HEC-RAS study Bitter Creek Trib14.prj: Bitter Creek Trib14 Base Level Engineering

--- Bitter Creek Trib14.g01 (geometry) --- (continued)

Type RM Length L Ch R = 1 ,34238   ,497,497,497
BEGIN DESCRIPTION:
Bitter Creek Trib14 53.0
END DESCRIPTION:
XS GIS Cut Line= 3
      1398154.97      6826587.99      1398653.78       6826748.5
      1398954.99      6826588.01
#Sta/Elev= 30
    4476 2300.31  4477.7 2300.31  4511.5  2299.4  4529.4 2299.62  4561.5 2294.49
  4588.3 2284.19  4633.6 2274.15  4738.7 2268.67    4786 2260.21  4830.8 2257.81
  4882.3 2249.44  4938.2 2246.86  4946.4 2241.52  4951.7 2243.98  4959.3 2237.26
  4975.5  2235.8    4976  2235.3  4992.1  2235.8    4998 2250.01  5009.4 2254.34
    5015 2253.05  5031.3 2259.27    5037 2255.44  5053.3 2259.88    5059 2256.72
  5075.3 2259.36  5097.2 2255.57  5171.3 2265.54  5185.1  2263.9  5341.3 2269.08
#Mann= 6 ,-1 , 0
    4476     .07       0  4477.7    .035       0  4511.5     .07       0
  4830.8     .16       0  4975.5     .07       0  4992.1     .07       0
Bank Sta=4975.5,4992.1
XS Rating Curve= 0 ,0
Exp/Cntr=0.3,0.1

Type RM Length L Ch R = 1 ,33741   ,498,498,498
BEGIN DESCRIPTION:
Bitter Creek Trib14 52.0
END DESCRIPTION:
XS GIS Cut Line= 3
      1398154.97      6826637.97      1398755.23      6827212.93
      1399746.22      6827247.52
#Sta/Elev= 30
  4168.8 2300.28  4218.4 2298.94  4296.1 2275.31  4345.7 2269.71    4565 2267.38
  4656.8 2261.53    4664 2258.73  4728.6 2255.99  4784.2 2253.75  4826.6 2247.66
  4918.4 2241.34  4960.4 2234.01  4966.6 2232.24  4967.1 2231.74  4983.5 2232.24
  4989.2  2233.8  4996.4 2241.14  5003.4 2241.73  5009.8 2248.73  5019.8 2250.17
  5039.8 2248.72  5089.8 2238.65  5099.8 2247.88  5119.8 2255.04  5149.9 2261.18
  5209.9  2259.2  5239.9 2253.53  5286.9 2261.76    5390 2270.95  5991.6 2296.78
#Mann= 5 ,-1 , 0
  4168.8     .07       0  4728.6     .16       0  4960.4     .07       0
  4966.6     .07       0  4983.5     .07       0
Bank Sta=4966.6,4983.5
XS Rating Curve= 0 ,0
Exp/Cntr=0.3,0.1

Type RM Length L Ch R = 1 ,33243   ,495,495,495
BEGIN DESCRIPTION:
Bitter Creek Trib14 51.0
END DESCRIPTION:
XS GIS Cut Line= 3
        1398355.        6827388.      1398471.43      6827571.23
      1398705.03        6827588.
#Sta/Elev= 30
  4782.9 2262.75  4863.4 2262.44  4905.7  2260.6    4921 2259.08  4926.9 2257.82
  4936.2 2257.58  4942.1  2253.8  4948.8  2255.6  4957.4 2256.31  4963.3 2252.24
  4972.5 2251.16  4978.5 2246.57  4984.5 2231.24  4990.2 2228.79  4990.7 2228.29
  5007.1 2228.79  5013.6 2232.25  5026.7 2232.09  5033.7 2232.84  5043.7  2235.2
  5063.7 2242.01  5103.8 2242.51  5113.9 2248.09    5154 2263.06  5161.7 2268.68
  5166.7 2268.62    5174 2273.12  5194.1 2281.91  5214.1 2288.48  5234.2 2290.48
#Mann= 3 ,-1 , 0
  4782.9     .07       0  4990.2     .07       0  5007.1     .07       0
Bank Sta=4990.2,5007.1
XS Rating Curve= 0 ,0
Exp/Cntr=0.3,0.1

Type RM Length L Ch R = 1 ,32748   ,497,497,497
BEGIN DESCRIPTION:
Bitter Creek Trib14 50.0
END DESCRIPTION:
XS GIS Cut Line= 3
      1398354.96      6827937.98       1398546.9      6828031.93
      1398755.03      6827837.97
#Sta/Elev= 30
  4786.3 2258.35  4817.3 2258.97  4867.9 2257.75  4929.9 2253.28  4935.4 2253.73
  4952.4 2243.72  4957.9 2239.42  4964.5 2228.29  4966.4 2227.24  4966.9 2226.74
  4983.3 2227.24  5002.1 2228.91  5008.7 2232.55  5015.5 2232.39  5022.8  2234.6
  5072.2 2240.97  5079.4 2243.08  5093.2 2244.85  5100.5 2247.13  5107.4  2247.5
  5114.7 2249.52  5157.2 2254.23    5164 2257.21  5171.4 2258.82  5206.5 2263.62
  5213.9 2265.59    5228 2271.66  5256.4 2279.52  5270.5 2282.05  5284.5  2282.4
#Mann= 3 ,-1 , 0
  4786.3     .07       0  4966.4     .07       0  4983.3     .07       0
Bank Sta=4966.4,4983.3
XS Rating Curve= 0 ,0
Exp/Cntr=0.3,0.1

Type RM Length L Ch R = 1 ,32251   ,499,499,499
BEGIN DESCRIPTION:
Bitter Creek Trib14 49.0
END DESCRIPTION:
XS GIS Cut Line= 3
        1398505.        6828438.      1398724.78      6828458.09
      1398854.98      6828188.04
#Sta/Elev= 30
  4779.3 2254.22  4839.6 2254.85  4889.8 2254.18  4919.9 2251.62  4944.5 2247.27
    4950 2243.27  4960.1  2239.7  4970.1 2234.27  4980.1 2227.78  5005.9 2226.06
  5006.4 2225.56  5022.8 2226.06  5031.4 2227.21    5037 2229.39  5066.7 2230.88
  5082.2 2233.66  5088.9 2235.77  5099.3 2235.92  5104.8 2237.15  5121.9 2238.57
  5133.3 2241.66  5188.8 2251.74    5211 2253.05  5233.2  2255.8  5246.1 2259.16
  5255.4 2260.39  5268.7 2264.67  5285.8 2268.29  5291.3 2270.95  5299.8 2271.92
#Mann= 3 ,-1 , 0
  4779.3     .07       0  5005.9     .07       0  5022.8     .07       0
Bank Sta=5005.9,5022.8
XS Rating Curve= 0 ,0
Exp/Cntr=0.3,0.1

Type RM Length L Ch R = 1 ,31752   ,498,498,498
BEGIN DESCRIPTION:
Bitter Creek Trib14 48.0
END DESCRIPTION:
XS GIS Cut Line= 3
      1398905.03      6828687.99      1399106.04      6828622.52
      1399305.04      6828688.01
#Sta/Elev= 30
  4788.6 2252.69  4820.1 2252.28  4862.2 2246.98  4868.4 2244.03  4914.8 2230.77
  4925.3 2230.47  4932.2 2231.54  4937.5 2229.87  4956.8 2226.94  4977.9 2227.24
  4988.4 2225.92  4990.7 2221.94  4991.2 2221.44  5007.7 2221.94    5020 2222.39
  5029.4 2226.67  5034.6 2222.26    5041 2235.64  5051.5 2253.57  5061.2 2258.18
  5066.4 2257.28  5072.6 2258.77  5092.9 2259.14    5130 2263.85  5135.8 2265.83
  5156.5 2268.03  5161.8  2267.5  5193.6 2269.81  5206.8 2273.48  5209.5 2273.48
#Mann= 3 ,-1 , 0
  4788.6     .07       0  4990.7     .07       0  5007.7     .07       0
Bank Sta=4990.7,5007.7
XS Rating Curve= 0 ,0
Exp/Cntr=0.3,0.1

Type RM Length L Ch R = 1 ,31254   ,498,498,498
BEGIN DESCRIPTION:
Bitter Creek Trib14 47.0
END DESCRIPTION:
XS GIS Cut Line= 3
      1398905.03      6828938.03      1399054.84      6829072.94
      1399254.97      6828988.01
#Sta/Elev= 30
  4798.4 2248.85  4852.2 2245.41  4876.5 2242.58  4904.9 2237.19  4911.6 2237.94
  4919.1  2236.1  4925.8 2236.46    4940 2232.97  4960.9 2231.09  4968.4 2229.12
  4976.6 2228.49  4989.3 2226.83  4996.7 2224.79  5002.8 2224.79    5011 2217.36
  5017.9 2216.69  5018.4 2216.19  5034.9 2216.69  5043.6 2222.87  5065.3 2223.35
  5073.7 2222.59  5097.4 2224.82  5102.8 2224.57  5108.8 2227.37  5119.7 2229.01
  5141.4 2236.24  5155.6 2242.33  5163.1 2248.97  5179.2 2254.96  5217.4 2263.12
#Mann= 5 ,-1 , 0
  4798.4     .07       0  4852.2     .16       0  4976.6     .07       0
  5017.9     .07       0  5034.9     .07       0
Bank Sta=5017.9,5034.9
XS Rating Curve= 0 ,0
Exp/Cntr=0.3,0.1

Type RM Length L Ch R = 1 ,30756   ,450,450,450
BEGIN DESCRIPTION:
Bitter Creek Trib14 46.0
END DESCRIPTION:
XS GIS Cut Line= 3
      1398405.04      6829388.01      1398955.33      6829538.14
      1399155.03      6829487.99
#Sta/Elev= 30
  4429.6 2268.65  4481.4 2256.24  4521.1  2251.5  4600.6 2245.66  4616.1 2242.16
  4714.6 2236.94  4788.8 2227.32  4823.4 2228.39  4828.6 2232.05  4854.5 2237.61
  4875.3  2238.8  4902.8 2232.47  4947.8 2226.98  4977.1 2217.67  4988.5 2216.91
    4989 2216.41  5005.9 2216.91  5059.3 2225.31  5064.4 2223.45  5082.1 2226.47
  5100.4 2232.86  5105.6 2229.32  5123.4 2235.89  5141.6 2239.35  5146.7 2235.11
  5164.6 2234.78  5174.9 2236.58  5182.7 2242.15  5195.6 2246.07  5205.9 2246.43
#Mann= 3 ,-1 , 0
  4429.6     .07       0  4988.5     .07       0  5005.9     .07       0
Bank Sta=4988.5,5005.9
XS Rating Curve= 0 ,0
Exp/Cntr=0.3,0.1

Type RM Length L Ch R = 1 ,30306   ,495,495,495
BEGIN DESCRIPTION:
Bitter Creek Trib14 45.0
END DESCRIPTION:
XS GIS Cut Line= 3
      1398605.03        6829888.      1398824.71      6829917.85
      1399005.04      6830038.02
#Sta/Elev= 30
  4778.3 2239.67  4798.5 2238.79  4814.5 2236.08  4819.5 2236.44  4838.8 2230.95
  4848.9 2231.54  4879.2 2231.21    4887 2230.48    4892 2226.45  4909.5    2225
    4970 2217.72  5003.2  2217.8  5007.8  2215.7  5013.8 2216.11  5019.9  2214.1
  5020.4  2213.6  5037.9  2214.1  5043.9 2224.08  5058.9 2229.39  5064.9 2227.24
  5079.9 2230.55  5085.9 2229.15    5101 2231.17    5116 2232.09    5131 2235.09
    5137 2234.15  5144.6 2238.07  5152.1 2238.04  5167.1 2239.55  5216.7 2239.73
#Mann= 3 ,-1 , 0
  4778.3     .07       0  5019.9     .07       0  5037.9     .07       0
Bank Sta=5019.9,5037.9
XS Rating Curve= 0 ,0
Exp/Cntr=0.3,0.1

Type RM Length L Ch R = 1 ,29811   ,497,497,497
BEGIN DESCRIPTION:
Bitter Creek Trib14 44.0
END DESCRIPTION:
XS GIS Cut Line= 3
      1398404.95      6830237.98      1398655.16      6830353.06
      1398854.99        6830338.
#Sta/Elev= 30
  4724.6 2238.09  4756.4 2234.14  4761.9 2234.81  4779.3 2232.54  4784.8 2233.01
  4790.7  2231.6  4813.3 2229.24  4853.7 2226.21  4889.8 2221.25  4899.7 2220.91
  4911.8 2219.29  4928.2 2218.15  4944.8 2218.17  4966.8 2217.03  4979.6 2215.57
  4988.8  2212.8  4990.9 2210.63  4991.4 2210.13  5008.4 2210.13  5008.9 2210.63
  5009.9 2212.21    5040 2214.99    5070 2220.21  5090.1 2221.99  5110.2 2225.26
  5129.5 2232.22  5134.6 2231.42  5160.3 2232.11  5190.4 2237.21  5200.4 2237.39
#Mann= 3 ,-1 , 0
  4724.6     .07       0  4990.9     .07       0  5008.9     .07       0
Bank Sta=4990.9,5008.9
XS Rating Curve= 0 ,0
Exp/Cntr=0.3,0.1

Type RM Length L Ch R = 1 ,29314   ,489,489,489
BEGIN DESCRIPTION:
Bitter Creek Trib14 43.0
END DESCRIPTION:
XS GIS Cut Line= 3
      1398009.82      6830686.56      1398421.78       6830771.4
      1398604.99        6830688.
#Sta/Elev= 30
  4579.4 2236.73  4756.6 2234.01  4819.5 2234.23  4857.2 2231.95  4862.3 2232.44
    4891 2229.62  4901.2 2229.89  4907.5 2228.64  4921.6 2222.77  4931.8 2220.08
  4962.9 2209.14  4972.7 2205.54  4973.9 2203.68  4974.4 2203.18  4991.9 2203.68
  4993.1 2205.89  4999.1 2209.23  5004.5 2209.23  5020.2  2214.2  5025.6  2213.7
  5043.2 2215.96  5058.5 2215.57  5089.3 2218.99  5094.8 2218.05  5102.4 2218.46
  5112.4 2219.96  5117.9 2219.77  5124.4 2221.53  5169.5 2224.42  5201.3 2228.58
#Mann= 3 ,-1 , 0
  4579.4     .07       0  4973.9     .07       0  4991.9     .07       0
Bank Sta=4973.9,4991.9
XS Rating Curve= 0 ,0
Exp/Cntr=0.3,0.1

Type RM Length L Ch R = 1 ,28825   ,497,497,497
BEGIN DESCRIPTION:
Bitter Creek Trib14 42.0
END DESCRIPTION:
XS GIS Cut Line= 3
      1398505.03      6831287.96      1398648.92      6831140.55
      1398804.97      6830988.03
#Sta/Elev= 30
    4794 2228.18  4845.3 2228.41  4864.6  2228.5  4892.9 2226.76    4900 2227.34
    4907 2225.43  4914.2 2225.18  4921.2 2222.98  4928.3 2222.22  4935.3 2219.78
  4942.5 2218.97  4949.5 2215.17  4956.6 2212.89  4963.6 2207.93  4970.8 2206.55
  4975.9 2203.02  4976.4 2202.52  4993.9 2203.02  4998.6 2204.52  5020.3 2208.48
  5034.4  2209.5    5091 2211.11  5112.2 2212.92  5147.6 2218.99  5182.9  2223.2
    5190 2223.18    5197 2225.44  5204.2 2226.46  5211.2 2229.64  5218.2 2229.01
#Mann= 5 ,-1 , 0
    4794     .07       0  4845.3    .035       0  4975.9     .07       0
  4993.9    .035       0  4998.6     .07       0
Bank Sta=4975.9,4993.9
XS Rating Curve= 0 ,0
Exp/Cntr=0.3,0.1

Type RM Length L Ch R = 1 ,28328   ,496,496,496
BEGIN DESCRIPTION:
Bitter Creek Trib14 41.0
END DESCRIPTION:
XS GIS Cut Line= 3
        1398605.        6831538.      1398809.19      6831539.73
      1398954.97      6831687.97
#Sta/Elev= 30
  4795.8 2224.93  4845.8 2220.83  4875.8 2215.98  4895.8 2210.68  4925.8 2208.39
  4945.8 2208.75  4975.8 2205.38  4985.8 2203.85  4993.8 2199.61  4994.3 2199.11
  5011.9 2199.61    5017 2202.27  5031.2 2203.82  5045.3 2203.91  5087.7 2210.65
  5094.9 2210.09  5101.9  2213.6    5109 2215.22    5116 2218.45  5123.1 2220.33
  5130.2 2224.98  5137.3 2225.59  5144.3 2231.01  5151.4 2231.79  5158.4 2239.78
  5165.6 2241.47  5172.6 2246.73  5179.7  2247.3  5193.9  2245.8  5207.9 2243.08
#Mann= 3 ,-1 , 0
  4795.8     .07       0  4993.8     .07       0  5011.9     .07       0
Bank Sta=4993.8,5011.9
XS Rating Curve= 0 ,0
Exp/Cntr=0.3,0.1

Type RM Length L Ch R = 1 ,27832   ,496,496,496
BEGIN DESCRIPTION:
Bitter Creek Trib14 40.0
END DESCRIPTION:
XS GIS Cut Line= 3
      1398504.97      6831887.99       1398691.1      6831974.84
      1398904.98      6831838.01
#Sta/Elev= 30
  4794.6 2224.97  4854.5  2224.8  4871.9 2223.31  4900.3 2217.68  4905.8 2218.51
  4923.1 2214.15  4928.6 2214.22  4938.1 2210.41    4946 2205.24  4951.5 2207.87
  4968.8 2197.67  4973.2  2197.1  4973.7  2196.6  4991.3  2197.1  4991.7 2197.74
  4997.2 2197.47  4999.4  2198.5  5022.2 2200.49  5028.4 2202.97  5037.4 2203.96
  5087.7 2205.38  5152.4 2209.92  5173.6 2209.78  5194.7 2212.02    5210 2214.29
  5218.3 2220.51  5231.1 2222.93  5240.4 2226.48  5246.3 2225.12  5253.9 2226.23
#Mann= 3 ,-1 , 0
  4794.6     .07       0  4973.2     .07       0  4991.3     .07       0
Bank Sta=4973.2,4991.3
XS Rating Curve= 0 ,0
Exp/Cntr=0.3,0.1

Type RM Length L Ch R = 1 ,27336   ,498,498,498
BEGIN DESCRIPTION:
Bitter Creek Trib14 39.0
END DESCRIPTION:
XS GIS Cut Line= 3
      1398704.96      6832438.01      1398903.68      6832398.55
      1399104.98      6832338.01
#Sta/Elev= 30
  4797.4 2219.74  4838.2 2219.45  4848.4 2218.06  4868.8 2214.24  4889.2 2207.16
  4909.6 2202.67  4930.4 2200.28  4940.2 2198.05  4950.4 2197.08  4967.4 2193.99
  4967.9 2193.49  4985.5 2193.99  5003.3 2195.35  5011.8 2196.91  5018.1  2200.3
  5023.4 2198.98  5032.7 2201.06  5043.1 2202.11  5051.2 2202.55  5056.4 2201.63
  5084.2 2203.92  5105.8 2206.61  5116.2 2206.65  5122.4 2208.17  5127.7 2207.82
  5147.6 2210.25  5155.5 2210.23  5188.5 2215.81  5199.8 2218.93  5210.2 2219.48
#Mann= 3 ,-1 , 0
  4797.4     .07       0  4967.4     .07       0  4985.5     .07       0
Bank Sta=4967.4,4985.5
XS Rating Curve= 0 ,0
Exp/Cntr=0.3,0.1

Type RM Length L Ch R = 1 ,26838   ,995,995,995
BEGIN DESCRIPTION:
Bitter Creek Trib14 38.0
END DESCRIPTION:
XS GIS Cut Line= 3
      1398005.04      6833187.99      1399185.21      6832767.91
      1399404.98        6832738.
#Sta/Elev= 30
  3747.3 2251.58  3788.2  2247.1  3793.5 2245.25    3819 2244.43  3824.3  2241.9
  3849.9    2241    3864 2237.95  3906.2  2234.2  3917.1 2231.46  4091.2 2220.85
  4161.2 2218.08  4419.8 2215.57  4717.5 2215.17  4773.8 2212.41    4810 2204.85
  4838.5 2202.74    4883 2199.42    4928 2198.83  4944.7  2195.3  4969.5 2190.68
    4970 2190.18  4987.6 2190.68  4997.2 2197.75  5002.4 2197.75  5009.9 2203.77
  5035.8 2209.83  5100.7 2217.65  5151.2 2228.73  5191.5 2230.53  5221.8 2227.99
#Mann= 5 ,-1 , 0
  3747.3     .07       0  4838.5     .16       0  4944.7     .07       0
  4969.5     .07       0  4987.6     .07       0
Bank Sta=4969.5,4987.6
XS Rating Curve= 0 ,0
Exp/Cntr=0.3,0.1

Type RM Length L Ch R = 1 ,25843   ,498,498,498
BEGIN DESCRIPTION:
Bitter Creek Trib14 37.0
END DESCRIPTION:
XS GIS Cut Line= 3
      1399304.98        6833638.      1399503.43       6833598.7
        1399555.      6833137.98
#Sta/Elev= 30
  4797.7 2208.42  4858.9 2208.83  4920.1 2207.75  4925.8  2204.1  4930.9 2207.79
  4940.4 2198.56  4950.6  2191.5  4960.8 2187.88    4977  2186.2  4982.4 2184.95
  4982.9 2184.45    5000 2184.45  5000.5 2184.95  5010.8 2187.95  5020.8  2189.9
    5041  2192.8  5090.2 2193.26  5111.4 2194.02  5131.5 2193.45  5141.6 2194.47
  5152.8 2194.29  5161.7 2193.14  5171.8 2194.03  5181.8 2193.26  5222.1 2194.67
  5232.1 2196.09  5252.3 2197.34  5292.5 2197.32  5444.5 2208.33  5463.6 2209.25
#Mann= 5 ,-1 , 0
  4797.7     .07       0  4982.4     .07       0  5000.5     .07       0
  5090.2     .16       0  5444.5     .07       0
Bank Sta=4982.4,5000.5
XS Rating Curve= 0 ,0
Exp/Cntr=0.3,0.1

Type RM Length L Ch R = 1 ,25345   ,488,488,488
BEGIN DESCRIPTION:
Bitter Creek Trib14 36.0
END DESCRIPTION:
XS GIS Cut Line= 3
      1399604.96      6833738.03      1399821.67      6833554.47
        1399855.      6833338.02
#Sta/Elev= 30
    4716 2204.62  4737.5 2203.49    4744 2203.93  4780.3 2203.08  4786.9  2200.9
  4794.6 2201.32  4801.2 2198.12  4807.8 2198.91  4815.5 2198.72    4822 2197.25
  4829.8 2197.04  4836.3 2195.87  4893.5 2190.66  4907.8 2191.04    4922 2190.52
  4936.3 2191.31  4964.9 2187.74  4992.3 2182.37  4997.4 2182.11  4997.9 2181.61
  5015.1 2181.61  5015.6 2182.11  5016.7 2185.85  5026.8 2193.39  5036.9 2195.72
  5067.2 2197.54  5077.4 2199.19  5116.6 2201.25    5128 2202.88    5219 2204.99
#Mann= 3 ,-1 , 0
    4716     .07       0  4997.4     .07       0  5015.6     .07       0
Bank Sta=4997.4,5015.6
XS Rating Curve= 0 ,0
Exp/Cntr=0.3,0.1

Type RM Length L Ch R = 1 ,24857   ,460,460,460
BEGIN DESCRIPTION:
Bitter Creek Trib14 35.0
END DESCRIPTION:
XS GIS Cut Line= 3
      1399704.96        6833988.      1400054.89      6833948.05
      1400254.98      6833688.02
#Sta/Elev= 30
  4647.8 2202.55  4657.9 2201.14    4678 2200.97  4698.2 2198.15  4728.8 2195.86
  4798.8 2192.45    4829 2193.24  4889.4 2191.45  4919.6  2187.9  4946.8 2186.97
  4969.9  2186.8  4997.5 2179.59  5012.6 2179.32  5013.1 2178.82  5031.2 2179.32
  5036.4  2182.3  5042.7 2188.37  5050.5 2187.62  5063.5 2192.98  5071.7 2192.91
    5078 2195.75  5086.2 2195.23  5092.5 2198.01  5156.9 2204.67  5235.7  2209.1
  5264.7  2213.9  5291.9 2223.29  5300.1 2224.61  5306.4 2227.37  5328.1 2231.44
#Mann= 5 ,-1 , 0
  4647.8     .07       0  4728.8     .16       0  4946.8     .07       0
  5012.6     .07       0  5031.2     .07       0
Bank Sta=5012.6,5031.2
XS Rating Curve= 0 ,0
Exp/Cntr=0.3,0.1

Type RM Length L Ch R = 1 ,24397   ,498,498,498
BEGIN DESCRIPTION:
Bitter Creek Trib14 34.0
END DESCRIPTION:
XS GIS Cut Line= 3
      1399804.99        6834438.      1400099.25      6834390.33
      1400454.97        6834438.
#Sta/Elev= 30
  4701.9 2200.92  4730.2 2199.23  4735.3 2199.73  4796.9 2192.32  4843.7    2185
  4934.9 2185.62    4945 2183.66  4955.2 2180.36  4965.3    2180  4972.6 2176.49
  4973.1 2175.99  4991.2 2176.49    5000 2176.78  5015.5 2185.05  5020.5 2185.38
    5026 2190.64  5036.1 2193.73  5038.9 2193.63  5056.2 2192.78  5098.5 2193.29
  5116.8    2195  5166.4 2197.62  5171.5  2197.3  5187.4 2199.14  5197.5 2198.63
  5217.7 2200.21  5249.5 2205.29  5328.7 2222.02  5338.7 2223.47  5358.9 2224.81
#Mann= 4 ,-1 , 0
  4701.9     .16       0  4972.6     .07       0  4991.2     .16       0
  5038.9     .07       0
Bank Sta=4972.6,4991.2
XS Rating Curve= 0 ,0
Exp/Cntr=0.3,0.1

Type RM Length L Ch R = 1 ,23899   ,484,484,484
BEGIN DESCRIPTION:
Bitter Creek Trib14 33.0
END DESCRIPTION:
XS GIS Cut Line= 3
      1399855.02        6834788.      1400054.66      6834838.37
      1400455.02      6834637.99
#Sta/Elev= 30
  4794.1 2198.89  4835.3 2199.39  4866.3 2197.65  4907.5 2197.63  4917.8 2195.51
  4928.2 2190.84  4935.2 2181.71  4940.4 2184.04  4948.8  2177.5  4960.1 2173.35
  4960.6 2172.85  4978.7 2173.35  5016.6  2178.9  5036.9 2180.28  5067.5 2177.79
  5098.4 2182.13  5112.2 2180.58  5148.7  2182.9  5193.4 2181.15  5232.5 2182.75
  5238.1 2184.83  5246.4 2184.47  5260.5 2187.29  5277.2 2188.08  5349.9 2199.74
  5394.4 2211.48  5411.4  2219.2  5416.9 2219.15  5433.7 2224.49  5447.7 2226.06
#Mann= 5 ,-1 , 0
  4794.1     .07       0  4960.1     .07       0  4978.7     .07       0
  5016.6     .16       0  5394.4     .07       0
Bank Sta=4960.1,4978.7
XS Rating Curve= 0 ,0
Exp/Cntr=0.3,0.1

Type RM Length L Ch R = 1 ,23415   ,474,474,474
BEGIN DESCRIPTION:
Bitter Creek Trib14 32.0
END DESCRIPTION:
XS GIS Cut Line= 3
        1400155.        6835038.      1400465.11      6834897.85
        1400455.        6834688.
#Sta/Elev= 30
  4659.7 2194.12  4691.6 2192.68  4714.6 2190.07  4725.7 2187.78  4743.3 2187.31
  4780.4 2182.54  4802.4 2181.06  4846.8 2180.66  4864.4 2179.32  4869.9 2180.17
  4901.1 2180.41  4923.1 2179.21    4956 2178.91  4977.9 2175.79  4987.9 2172.42
  4988.4 2171.92  5006.5 2172.42  5039.9 2175.94  5049.9 2180.24  5052.9 2182.62
  5059.9 2188.18  5069.9 2193.27    5100 2195.98  5105.6 2197.94  5110.6 2197.85
    5130    2202    5150 2206.86  5178.6    2218  5190.1 2221.21  5210.1 2223.58
#Mann= 5 ,-1 , 0
  4659.7     .07       0  4987.9     .07       0  5006.5     .07       0
  5052.9     .16       0  5178.6     .07       0
Bank Sta=4987.9,5006.5
XS Rating Curve= 0 ,0
Exp/Cntr=0.3,0.1

Type RM Length L Ch R = 1 ,22941   ,399,399,399
BEGIN DESCRIPTION:
Bitter Creek Trib14 31.0
END DESCRIPTION:
XS GIS Cut Line= 3
      1400205.03        6835238.      1400541.63      6835274.68
        1400955.        6834838.
#Sta/Elev= 30
  4661.4 2192.76  4889.9 2189.45  4912.9 2189.91  4922.9  2187.4    4943 2172.46
  4953.9 2170.07  4954.4 2169.57  4972.5 2170.07  4981.4 2172.11  4986.4 2171.37
  5007.2  2173.2  5014.1  2172.6  5021.4 2176.47  5028.3  2177.2  5056.6 2176.55
  5120.1 2178.03  5155.7 2181.04  5162.6 2180.53  5169.9 2182.05  5190.9 2181.53
  5233.4 2183.08    5269 2186.09  5346.6 2190.18  5509.3 2194.42  5537.6 2197.29
  5552.5 2200.89  5560.4 2202.62  5580.1 2209.17  5597.9 2213.73  5601.3 2213.73
#Mann= 5 ,-1 , 0
  4661.4     .07       0  4953.9     .07       0  4972.5     .07       0
  5552.5     .16       0  5560.4     .07       0
Bank Sta=4953.9,4972.5
XS Rating Curve= 0 ,0
Exp/Cntr=0.3,0.1

Type RM Length L Ch R = 1 ,22542   ,565,565,565
BEGIN DESCRIPTION:
Bitter Creek Trib14 30.0
END DESCRIPTION:
XS GIS Cut Line= 3
      1400505.03      6835787.98      1400849.97      6835488.81
      1400999.36        6835209.
#Sta/Elev= 30
  4543.4 2187.42  4621.7 2186.65  4628.4 2187.38    4806 2187.18  4841.1  2186.3
  4954.1 2180.88  4961.7 2175.02    4976 2173.17  4982.6 2170.38  4990.2 2171.32
  4996.8 2169.04    5003 2168.08  5003.5 2167.58  5021.6 2168.08  5025.3  2169.6
  5034.9 2170.96  5079.8 2173.23  5085.5 2172.05  5091.6 2173.83  5123.7 2176.01
  5129.4 2174.82  5167.6 2176.18  5182.3 2177.93  5189.6 2179.86  5195.2 2179.72
  5211.5 2181.61  5217.2 2181.22  5227.6 2182.88  5271.7 2187.08  5317.2 2188.15
#Mann= 3 ,-1 , 0
  4543.4     .07       0    5003     .07       0  5021.6     .07       0
Bank Sta=5003,5021.6
XS Rating Curve= 0 ,0
Exp/Cntr=0.3,0.1

Type RM Length L Ch R = 1 ,21977   ,499,499,499
BEGIN DESCRIPTION:
Bitter Creek Trib14 29.0
END DESCRIPTION:
XS GIS Cut Line= 3
      1400905.02      6835937.98      1401255.12      6835677.95
      1401454.97      6835488.03
#Sta/Elev= 30
  4563.9 2184.44  4627.5 2183.71  4689.6 2181.17    4772 2178.93  4777.7 2177.61
  4900.2 2175.72  4936.3 2169.13  4942.5 2170.43  4957.1  2168.2  4963.3 2168.72
  4971.7 2166.74    4978 2167.94  4986.3  2165.1  4992.6  2165.4  4996.8 2163.37
  5003.4 2163.37  5004.5 2162.36    5005 2161.86  5023.2 2162.36    5028  2165.3
  5035.3 2171.53  5042.2 2170.66  5049.4 2176.83  5056.3 2173.57  5063.6 2176.41
  5070.5 2175.41  5077.7 2177.51  5155.4    2180    5212    2183  5275.7 2184.18
#Mann= 5 ,-1 , 0
  4563.9     .07       0  4689.6     .16       0    4772     .07       0
  5004.5     .07       0  5023.2     .07       0
Bank Sta=5004.5,5023.2
XS Rating Curve= 0 ,0
Exp/Cntr=0.3,0.1

Type RM Length L Ch R = 1 ,21478   ,458,458,458
BEGIN DESCRIPTION:
Bitter Creek Trib14 28.0
END DESCRIPTION:
XS GIS Cut Line= 3
      1401055.02        6836038.      1401454.59      6836043.17
      1401655.02        6836038.
#Sta/Elev= 30
  4600.4 2182.97  4740.4 2180.56  4820.4 2177.59  4850.4 2177.21  4860.4 2176.45
  4870.4 2174.69  4880.4 2174.43  4890.4 2175.14  4910.4 2175.02  4950.4 2170.55
  4960.4 2170.57  4970.4 2168.79  4980.4 2168.55  4986.1 2166.75  4991.1 2170.02
  4997.7 2164.82  5002.7 2164.82    5006 2161.24  5011.1 2160.58  5011.6 2160.08
  5029.8 2160.58  5030.4 2166.98  5060.4 2175.27  5070.4 2179.92  5080.4 2181.16
  5110.5 2179.41  5160.5 2182.24  5170.5 2186.94  5180.5 2189.87  5200.5 2193.13
#Mann= 3 ,-1 , 0
  4600.4     .07       0  5011.1     .07       0  5029.8     .07       0
Bank Sta=5011.1,5029.8
XS Rating Curve= 0 ,0
Exp/Cntr=0.3,0.1

Type RM Length L Ch R = 1 ,21020   ,500,500,500
BEGIN DESCRIPTION:
Bitter Creek Trib14 27.0
END DESCRIPTION:
XS GIS Cut Line= 3
      1401254.96      6836337.99      1401656.65      6836427.32
      1401754.98      6836238.03
#Sta/Elev= 30
  4588.5 2180.64  4607.7 2179.32    4705 2177.25  4748.6 2174.58  4753.7 2175.81
  4772.9 2173.55  4813.9 2171.74  4824.2 2169.78  4834.4 2169.04  4865.1 2168.06
  4927.5 2168.49  4948.9 2166.25  4967.6  2163.9  4976.4 2160.61  4978.7    2159
  4979.2  2158.5  4997.4    2159  5002.4 2159.33  5006.1  2160.8  5028.2  2162.4
  5033.8 2165.33  5050.3 2165.93  5055.9 2167.66  5072.4 2170.05  5078.1 2168.49
  5088.9 2168.28  5100.6  2172.9    5111 2176.06  5116.6 2175.75  5213.3 2179.29
#Mann= 5 ,-1 , 0
  4588.5     .07       0  4927.5     .16       0  4948.9     .07       0
  4978.7     .07       0  4997.4     .07       0
Bank Sta=4978.7,4997.4
XS Rating Curve= 0 ,0
Exp/Cntr=0.3,0.1

Type RM Length L Ch R = 1 ,20520   ,1691,1691,1691
BEGIN DESCRIPTION:
Bitter Creek Trib14 26.0
END DESCRIPTION:
XS GIS Cut Line= 3
      1401154.98      6837088.01      1401762.82      6836894.19
        1402355.        6836488.
#Sta/Elev= 30
    4362 2185.79  4442.5 2181.07  4456.5 2181.67  4474.7 2179.32  4576.6 2176.45
  4886.8 2174.89  4903.9 2172.86  4918.3 2172.55  4981.3 2164.33  4998.5 2157.85
  5004.3  2156.7  5004.8  2156.2  5024.2  2156.7  5026.9  2159.7  5035.2 2162.87
  5063.3 2166.88    5092 2166.54  5121.8 2164.68    5136 2165.77  5142.8 2168.82
  5157.7 2169.93  5184.1 2169.28  5372.9 2168.76  5402.7 2166.06  5414.9 2168.04
  5444.7 2168.95  5450.7  2170.1  5510.3 2174.37    5603 2183.55  5718.1 2191.12
#Mann= 5 ,-1 , 0
    4362     .07       0  5004.3     .07       0  5024.2     .07       0
  5184.1     .16       0  5450.7     .07       0
#XS Ineff= 2 , 0
                         5328.93         2175.58
Permanent Ineff=
       F       F
Bank Sta=5004.3,5024.2
XS Rating Curve= 0 ,0
Exp/Cntr=0.3,0.1

Type RM Length L Ch R = 1 ,18829   ,596,596,596
BEGIN DESCRIPTION:
Bitter Creek Trib14 25.0
END DESCRIPTION:
XS GIS Cut Line= 3
      1401855.02        6837338.      1402607.73      6837281.84
      1403005.02      6836687.98
#Sta/Elev= 30
  4245.2 2173.48  4278.5 2173.11  4357.9 2172.46  4562.1 2170.69  4676.4 2167.53
  4728.5 2164.98  4761.1 2164.02  4860.5 2163.63  4927.1 2162.89    4960 2158.01
  4967.2 2157.17  4977.2 2153.04  4978.3 2148.69  4978.8 2148.19  4998.4 2148.69
  5022.4 2156.14  5052.4 2158.54  5064.8 2158.47    5083 2161.43  5115.5 2166.01
    5137 2167.67  5198.6 2167.99  5310.6 2169.16  5382.7 2170.93  5541.8 2178.59
  5634.9 2186.95  5664.9 2191.82  5678.4 2200.22    5692 2203.74  5714.5 2204.08
#Mann= 12 ,-1 , 0
  4245.2     .07       0  4278.5    .035       0  4357.9     .07       0
  4562.1    .035       0  4728.5     .07       0  4761.1    .035       0
  4860.5     .16       0    4960     .07       0  4978.3     .07       0
  4998.4     .07       0    5083     .16       0  5198.6     .07       0
Bank Sta=4978.3,4998.4
XS Rating Curve= 0 ,0
Exp/Cntr=0.3,0.1

Type RM Length L Ch R = 1 ,18233   ,1739,1739,1739
BEGIN DESCRIPTION:
Bitter Creek Trib14 24.0
END DESCRIPTION:
XS GIS Cut Line= 3
      1401304.97      6839288.03      1402928.18      6837761.71
      1403155.02      6837387.97
#Sta/Elev= 30
  2771.9 2207.51  2979.3 2195.73  3173.5 2183.89  3429.5 2173.03  3712.9 2166.59
  3903.8 2166.77  3932.2    2164  3962.3 2165.84  3988.8 2164.29  4009.8 2165.53
  4377.9 2162.47  4611.3 2164.87  4844.6 2164.42  4908.5 2161.24    4972 2154.11
  4999.1 2153.79    5016 2149.78  5018.1 2144.97  5018.6 2144.47  5038.3 2144.97
  5043.7 2151.93  5051.1 2154.52  5101.8  2156.2  5117.3  2158.4  5123.2 2157.05
  5196.8 2157.56    5255 2160.09  5313.1 2165.36  5349.9 2171.12  5437.2 2177.02
#Mann= 7 ,-1 , 0
  2771.9     .07       0  2979.3    .035       0  3173.5     .07       0
  3429.5    .035       0  3962.3     .07       0  5018.1     .07       0
  5038.3     .07       0
Bank Sta=5018.1,5038.3
XS Rating Curve= 0 ,0
Exp/Cntr=0.3,0.1

Type RM Length L Ch R = 1 ,16494   ,421,421,421
BEGIN DESCRIPTION:
Bitter Creek Trib14 23.0
END DESCRIPTION:
XS GIS Cut Line= 3
      1402655.03      6839187.97      1404250.03      6837637.94
      1403882.28      6836964.96
#Sta/Elev= 30
  2775.9 2173.78  2896.8 2166.51  2973.8 2161.38    3112 2158.72  3346.5 2157.62
  3426.5 2159.02  3461.8 2155.56  3490.1  2157.9  3519.7 2156.53  4055.9 2157.24
  4494.8  2154.5  4501.1 2154.31  4529.7 2153.64  4572.2 2145.57  4854.9 2149.25
  4883.2 2147.22  4904.5 2148.71  4961.1 2145.75  4975.2 2143.34  4979.3 2139.17
  4979.8 2138.67  4999.5 2139.17  5040.8 2147.88  5056.9 2148.56  5062.6 2150.59
  5084.4 2149.29  5100.8 2152.39  5122.4 2155.34  5171.7 2156.74  5766.9 2165.73
#Mann= 10 ,-1 , 0
  2775.9     .07       0  2896.8    .035       0    3112     .07       0
  3346.5    .035       0  3519.7     .07       0  4494.8     .16       0
  4501.1     .07       0  4979.3     .07       0  4999.5     .07       0
  5100.8     .07       0
#XS Ineff= 2 , 0
         4742.13 2155.91
Permanent Ineff=
       F       F
Bank Sta=4979.3,4999.5
XS Rating Curve= 0 ,0
Exp/Cntr=0.3,0.1

Type RM Length L Ch R = 1 ,16073   ,652,652,652
BEGIN DESCRIPTION:
Bitter Creek Trib14 22.0
END DESCRIPTION:
XS GIS Cut Line= 3
      1402955.01      6839287.99      1404415.19      6837897.68
      1404905.01      6837387.99
#Sta/Elev= 30
  2983.8 2174.69  3171.3 2161.22  3365.6 2155.77  3457.6 2156.96  3549.8 2148.42
  3570.9 2149.11  3613.3 2159.31  3669.9  2152.9  3719.3 2151.35  3761.8  2155.1
  3790.1 2148.89    3809 2150.05  3832.6 2153.09    3875 2149.42  3938.5  2152.9
  4253.6 2152.74  4513.2  2152.2  4773.3 2151.23  4844.1 2144.34  4985.7 2147.22
  4992.6 2144.95  4996.1 2136.98  4996.6 2136.48  5017.3 2136.98  5077.5  2147.7
  5197.9 2147.12    5219 2140.82  5261.4 2148.89  5458.6 2158.12  5706.9 2171.92
#Mann= 10 ,-1 , 0
  2983.8    .035       0  3171.3     .07       0  3365.6    .035       0
    3809     .07       0  4253.6     .16       0  4513.2     .07       0
  4996.1     .07       0  5017.3     .07       0  5197.9     .16       0
  5458.6     .07       0
#XS Ineff= 2 , 0
         4123.86 2161.69
Permanent Ineff=
       F       F
Bank Sta=4996.1,5017.3
XS Rating Curve= 0 ,0
Exp/Cntr=0.3,0.1

Type RM Length L Ch R = 1 ,15421   ,504,504,504
BEGIN DESCRIPTION:
Bitter Creek Trib14 21.0
END DESCRIPTION:
XS GIS Cut Line= 4
      1403955.03      6839437.96      1404873.39      6837941.33
      1404870.34       6837838.8      1404830.94      6837565.83
#Sta/Elev= 30
  3141.5 2161.02    3155 2162.38  3207.2    2158  3301.9 2155.33    3708 2152.49
  3729.3 2151.01  3749.4 2152.52  3781.4 2150.82  4414.1 2146.99    4493 2146.16
  4529.7 2141.91  4545.1 2145.74  4645.9 2146.35  4676.6 2147.57    4784 2143.96
  4798.5 2145.31  4842.7 2143.16  4863.2 2144.35  4877.9 2143.21  4940.8 2145.03
  4960.8  2138.7  4970.8 2138.86  4980.2 2134.17  4980.7 2133.67  5001.4 2134.17
  5004.1 2136.29  5041.2 2143.87  5072.4 2148.42  5132.2  2155.9  5275.8 2161.33
#Mann= 8 ,-1 , 0
  3141.5    .035       0  3749.4     .07       0  4414.1     .16       0
  4645.9     .07       0  4863.2     .16       0  4980.2     .07       0
  5001.4     .16       0  5072.4     .07       0
#XS Ineff= 2 , 0
         4682.74  2150.6
Permanent Ineff=
       F       F
Bank Sta=4980.2,5001.4
XS Rating Curve= 0 ,0
Exp/Cntr=0.3,0.1

Type RM Length L Ch R = 1 ,14917   ,599,599,599
BEGIN DESCRIPTION:
Bitter Creek Trib14 20.0
END DESCRIPTION:
XS GIS Cut Line= 3
      1403955.01      6839637.99      1405104.91      6838108.04
        1405405.        6837838.
#Sta/Elev= 30
  3086.1 2181.64  3128.8 2179.13  3143.4 2175.55  3286.2 2163.78  3293.3 2161.52
  3312.5 2161.66  3493.3 2153.89  3923.9 2150.87  4449.6 2147.03  4466.6 2147.14
  4656.4 2145.25  4722.1 2138.36  4736.6 2144.34  4809.1 2145.07  4836.6 2145.19
  4878.3 2141.14  4936.6 2142.28    4972 2138.83  4978.2 2134.81  4986.6 2135.03
  4996.6  2131.2  4997.1  2130.7  5017.8  2131.2  5021.4 2133.46  5042.3 2135.53
  5049.8 2140.85  5056.5 2142.77  5113.3 2145.73  5148.5 2153.08  5403.7 2170.52
#Mann= 9 ,-1 , 0
  3086.1     .07       0  3312.5    .035       0  3923.9     .07       0
  4449.6     .16       0  4466.6     .07       0  4656.4     .16       0
  4809.1     .07       0  4996.6     .07       0  5017.8     .07       0
#XS Ineff= 2 , 0
         4814.72 2151.11
Permanent Ineff=
       F       F
Bank Sta=4996.6,5017.8
XS Rating Curve= 0 ,0
Exp/Cntr=0.3,0.1

Type RM Length L Ch R = 1 ,14318   ,598,598,598
BEGIN DESCRIPTION:
Bitter Creek Trib14 19.0
END DESCRIPTION:
XS GIS Cut Line= 3
      1403904.97      6839738.02      1405488.29      6838471.43
        1405505.      6837988.02
#Sta/Elev= 30
  2972.4 2187.31  3136.5 2183.39  3171.7 2180.43  3221.4  2172.9  3335.3 2164.85
  3341.1 2164.75  3444.2 2157.74  3727.2 2150.73  4074.6 2146.64  4088.9 2147.77
  4537.2 2144.34  4857.4 2144.04  4900.6 2142.28  4935.8 2137.53  4985.4  2138.9
  4993.4 2137.65    5002 2128.45  5002.5 2127.95  5024.8 2128.45  5043.5 2134.69
  5048.9 2139.46  5057.7 2140.01  5093.5  2138.2  5143.5 2139.53  5183.5  2145.7
  5223.6 2146.16  5293.6 2150.85  5313.6 2150.04  5343.1 2153.43  5483.7 2164.07
#Mann= 9 ,-1 , 0
  2972.4     .07       0  3335.3    .035       0  3341.1     .07       0
  3444.2    .035       0  4088.9     .07       0    5002     .07       0
  5024.8     .07       0  5057.7     .16       0  5343.1     .07       0
Bank Sta=5002,5024.8
XS Rating Curve= 0 ,0
Exp/Cntr=0.3,0.1

Type RM Length L Ch R = 1 ,13720   ,648,648,648
BEGIN DESCRIPTION:
Bitter Creek Trib14 18.0
END DESCRIPTION:
XS GIS Cut Line= 3
      1404505.01      6839587.99       1405964.7      6838798.76
        1406505.      6837987.99
#Sta/Elev= 30
  3340.6 2176.87  3370.6 2176.24  3396.1 2171.48  3414.3  2167.7  3442.9 2167.24
  3488.4 2159.87  3583.7 2153.65  3693.1 2148.95  3738.5    2150  3970.2 2145.79
  4071.5 2144.86  4267.4 2143.71  4714.1 2141.65  4852.5 2138.85  4920.8 2135.97
  4954.9 2128.72  4965.3 2128.73  4966.1 2126.33  4966.6 2125.83    4989 2126.33
  4997.3 2135.93  5057.8 2135.59  5080.3 2135.45  5101.4 2139.07  5116.4 2136.99
  5122.4 2139.92  5125.9 2139.12    5483 2146.69  5685.9 2158.62  5974.3 2170.45
#Mann= 9 ,-1 , 0
  3340.6     .07       0  3396.1    .035       0  3970.2     .07       0
  4071.5    .035       0  4267.4     .07       0  4966.1     .07       0
    4989     .07       0  5057.8     .16       0  5125.9     .07       0
Bank Sta=4966.1,4989
XS Rating Curve= 0 ,0
Exp/Cntr=0.3,0.1

Type RM Length L Ch R = 1 ,13072   ,265,265,265
BEGIN DESCRIPTION:
Bitter Creek Trib14 17.0
END DESCRIPTION:
XS GIS Cut Line= 4
       1405494.7      6839128.52        1405724.      6839172.14
      1406356.87      6839276.91       1407439.3      6839550.62
#Sta/Elev= 30
  4125.1 2142.29  4796.4 2139.08  4835.9 2133.12  4866.3 2132.78  4927.2 2135.24
  4957.6 2134.33  4967.7 2131.28  4974.4 2126.28  4979.5 2130.39    4985 2124.34
  4985.5 2123.84    5008 2124.34  5008.4 2125.59  5024.4 2131.43  5029.5    2131
  5039.3 2133.18  5049.6 2132.73  5116.3 2135.74  5163.1 2137.25  5217.7 2136.37
  5319.1 2135.46  5420.5 2135.18  5503.5 2136.11  5627.3  2135.1  5724.6 2130.17
  5757.6 2127.81  5792.3 2127.76  5914.1 2135.61  6050.2 2143.24  6116.5 2145.21
#Mann= 9 ,-1 , 0
  4125.1     .07       0    4985     .07       0    5008     .07       0
  5116.3     .16       0  5217.7     .07       0  5319.1     .16       0
  5420.5     .07       0  5724.6    .035       0  5914.1     .07       0
#XS Ineff= 2 , 0
                         5276.65         2139.88
Permanent Ineff=
       F       F
Bank Sta=4985,5008
XS Rating Curve= 0 ,0
Exp/Cntr=0.3,0.1

Type RM Length L Ch R = 1 ,12807   ,1364,1364,1364
BEGIN DESCRIPTION:
Bitter Creek Trib14 16.0
END DESCRIPTION:
XS GIS Cut Line= 4
        1405447.      6839323.84      1405668.11      6839369.41
      1406434.72      6839508.03      1407536.57      6839662.37
#Sta/Elev= 30
  3995.2 2142.89  4027.9 2142.32  4524.9 2139.68  4578.4 2137.31  4652.4 2138.26
  4675.1 2136.64  4729.2    2138  4759.7  2137.5  4919.8 2132.72  4939.3 2124.83
  4978.6 2123.83  4979.1 2123.33  5001.6 2123.83  5081.1 2132.35  5128.9 2132.79
  5228.4 2131.38  5272.9 2131.57  5303.2 2134.69  5505.2 2132.93  5606.1 2131.22
  5656.6 2128.76  5666.7  2125.3  5676.8 2127.97  5754.6 2130.79  5838.4 2131.13
  5968.8  2141.1  5973.8 2139.19  6024.9 2142.91  6070.6 2146.62  6112.6 2146.17
#Mann= 10 ,-1 , 0
  3995.2     .07       0  4027.9    .035       0  4652.4     .07       0
  4729.2    .035       0  4759.7     .07       0  4978.6     .07       0
  5001.6     .07       0  5128.9     .16       0  5228.4    .035       0
  6024.9     .16       0
#XS Ineff= 2 , 0
                         5351.78         2139.63
Permanent Ineff=
       F       F
Bank Sta=4978.6,5001.6
XS Rating Curve= 0 ,0
Exp/Cntr=0.3,0.1

Type RM Length L Ch R = 1 ,11443   ,594,594,594
BEGIN DESCRIPTION:
Bitter Creek Trib14 15.0
END DESCRIPTION:
XS GIS Cut Line= 3
      1405554.97      6840738.01      1407535.25      6839917.59
      1407856.76      6839401.43
#Sta/Elev= 30
  2856.5 2165.54  2958.4 2158.17  3107.8 2148.58  3116.3 2149.84  3258.9 2142.58
  3397.7 2136.83  3527.9 2134.37  3836.2 2131.83  4285.2 2131.77    4328 2130.16
  4362.7    2133  4404.9 2131.53  4490.6 2130.11  4573.4 2129.78  4794.1 2127.03
  4931.5 2118.39  4955.4 2120.69  4960.8 2126.66  4984.7 2126.45  4995.4 2116.79
  4995.9 2116.29    5019 2116.79  5022.5 2126.25  5034.9 2132.34  5058.4 2140.19
  5071.9 2141.86  5140.8 2142.75  5207.8 2141.93  5346.7 2140.08  5608.1 2145.97
#Mann= 13 ,-1 , 0
  2856.5     .07       0  2958.4    .035       0  3258.9     .07       0
  4285.2    .035       0  4404.9     .07       0  4490.6    .035       0
  4573.4     .16       0  4995.4     .07       0    5019     .16       0
  5071.9    .035       0  5140.8     .16       0  5207.8     .07       0
  5346.7    .035       0
Bank Sta=4995.4,5019
XS Rating Curve= 0 ,0
Exp/Cntr=0.3,0.1

Type RM Length L Ch R = 1 ,10849   ,570,570,570
BEGIN DESCRIPTION:
Bitter Creek Trib14 14.0
END DESCRIPTION:
XS GIS Cut Line= 3
      1405904.96      6840738.01      1407521.56       6840404.7
      1408204.96      6840288.01
#Sta/Elev= 30
  3349.4 2148.56    3466    2145  3575.7 2140.02  3890.6 2132.33  4454.1 2128.71
  4503.2 2127.16  4554.3 2130.65  4595.1  2127.9  4643.2 2128.33  4862.8 2128.98
    4908 2124.01  4983.1 2124.71  4993.3 2121.84  4997.5 2116.09    4998 2115.59
  5021.1 2116.09  5023.8  2122.5  5033.9 2124.14  5044.1 2119.31  5064.4 2124.66
  5196.2  2124.9  5287.5 2127.87    5305 2130.04  5409.3 2132.54  5449.9 2136.21
    5460 2135.32  5517.6 2138.94  5610.8 2142.54  5665.8 2144.07  5693.3 2147.52
#Mann= 8 ,-1 , 0
  3349.4    .035       0    3466     .07       0  4454.1    .035       0
  4643.2     .16       0  4997.5     .07       0  5021.1     .16       0
  5517.6     .07       0  5610.8    .035       0
#XS Ineff= 2 , 0
         4556.35 2134.16
Permanent Ineff=
       F       F
Bank Sta=4997.5,5021.1
XS Rating Curve= 0 ,0
Exp/Cntr=0.3,0.1

Type RM Length L Ch R = 1 ,10279   ,581,581,581
BEGIN DESCRIPTION:
Bitter Creek Trib14 13.0
END DESCRIPTION:
XS GIS Cut Line= 3
      1405505.03        6840788.      1407924.84      6840808.39
        1408305.        6840638.
#Sta/Elev= 30
  2580.1 2169.01  2692.4 2161.31  2820.1 2154.75  2935.2 2153.55  3122.8 2149.43
  3203.2 2145.49  3530.1  2138.9  3560.1 2137.81  3590.1 2133.03  3620.1 2134.48
  3680.1 2131.69  4000.1 2129.12  4070.1 2125.67  4084.3 2126.99  4120.1 2129.09
  4140.1  2126.6  4219.9 2126.09  4770.2 2124.94  4850.2 2121.16  5002.8 2121.29
  5014.9 2119.65  5020.7 2113.88  5021.2 2113.38  5044.4 2113.88    5055 2121.71
  5089.9 2119.65  5120.7 2126.94    5165 2131.86  5309.5 2142.65  5416.6 2146.47
#Mann= 9 ,-1 , 0
  2580.1     .07       0  2692.4    .035       0  2935.2     .07       0
  3122.8    .035       0  3203.2     .07       0  4084.3    .035       0
  4219.9     .16       0  5020.7     .07       0  5044.4     .16       0
Bank Sta=5020.7,5044.4
XS Rating Curve= 0 ,0
Exp/Cntr=0.3,0.1

Type RM Length L Ch R = 1 ,9698    ,599,599,599
BEGIN DESCRIPTION:
Bitter Creek Trib14 12.0
END DESCRIPTION:
XS GIS Cut Line= 3
      1406455.01        6840938.       1407904.3      6841167.85
      1408555.01        6841138.
#Sta/Elev= 30
  3532.6 2161.49  3561.2 2166.03  3566.3 2168.39  3583.2 2167.89  3623.5 2160.16
  3628.6 2164.65  3633.8 2161.63  3690.9 2146.25  3695.9 2147.75  3753.2 2138.86
  3897.1 2131.28  4024.3 2128.87  4210.4 2126.01  4471.3 2122.06  4655.8 2121.64
  4747.6 2122.96  4842.6 2121.58  4919.7 2123.85    4940  2120.3  4948.4 2111.83
  4948.9 2111.33  4972.1 2111.83  4980.5 2115.83  4997.8 2118.92  5130.8 2119.13
  5150.9 2120.69  5200.9 2119.43    5291 2123.55  5511.2 2142.52  5651.4 2158.07
#Mann= 7 ,-1 , 0
  3532.6     .07       0  4024.3    .035       0  4210.4     .16       0
  4471.3     .07       0  4655.8     .16       0  4948.4     .07       0
  4972.1     .16       0
Bank Sta=4948.4,4972.1
XS Rating Curve= 0 ,0
Exp/Cntr=0.3,0.1

Type RM Length L Ch R = 1 ,9099    ,599,599,599
BEGIN DESCRIPTION:
Bitter Creek Trib14 11.0
END DESCRIPTION:
XS GIS Cut Line= 3
      1406604.99        6841088.      1408213.51      6841634.43
      1408904.97      6841088.02
#Sta/Elev= 30
  3301.2 2152.37  3480.8 2137.52  3598.7 2131.73  3828.8 2125.89  3860.6 2125.93
  4089.8 2123.53  4424.5 2119.45  4619.3 2120.02  4642.5 2121.91  4718.7 2120.92
  4744.8 2117.72  4750.1 2119.33  4832.6  2115.9  4995.9 2117.65  5015.5 2110.21
    5016 2109.71  5039.3 2110.21  5040.5 2113.22    5063 2116.63  5176.8 2115.89
  5333.3 2129.49  5489.4 2147.45  5503.8 2149.64  5518.3 2154.86  5547.1 2158.78
  5599.1 2162.22  5689.8 2165.54  5771.3 2174.43  5851.9 2185.16  5881.3 2190.41
#Mann= 11 ,-1 , 0
  3301.2     .07       0  3598.7    .035       0  3828.8     .07       0
  3860.6     .16       0  4089.8     .07       0  4424.5     .16       0
  5015.5     .07       0  5039.3     .16       0  5599.1    .035       0
  5771.3     .16       0  5851.9     .07       0
Bank Sta=5015.5,5039.3
XS Rating Curve= 0 ,0
Exp/Cntr=0.3,0.1

Type RM Length L Ch R = 1 ,8500    ,547,547,547
BEGIN DESCRIPTION:
Bitter Creek Trib14 10.0
END DESCRIPTION:
XS GIS Cut Line= 3
        1406555.        6841238.      1408138.29      6841954.57
      1408504.98      6842137.99
#Sta/Elev= 30
  3262.1 2163.99  3338.9 2159.95  3466.7  2141.8  3582.6 2133.04  3764.9 2127.54
  4020.4 2126.11  4071.7 2125.46  4094.8 2121.16  4100.3 2124.78  4198.2 2126.26
  4289.6 2123.51  4388.5 2118.88  4408.5 2121.69  4607.4 2114.48  4676.7 2119.68
  4779.2 2114.84  4835.3 2114.32  4911.4 2115.72  4970.4 2115.52  4981.6 2108.67
  4982.1 2108.17  5005.4 2108.67  5021.6 2113.63  5092.1 2116.38  5150.3 2127.31
  5217.2 2132.95  5267.5 2132.58  5334.6 2141.89  5351.3 2147.55    5410 2149.01
#Mann= 13 ,-1 , 0
  3262.1     .07       0  3582.6    .035       0  3764.9     .07       0
  4020.4    .035       0  4289.6     .07       0  4408.5     .16       0
  4779.2     .12       0  4835.3     .16       0  4911.4     .12       0
  4981.6     .07       0  5005.4     .12       0  5092.1     .16       0
  5150.3    .035       0
Bank Sta=4981.6,5005.4
XS Rating Curve= 0 ,0
Exp/Cntr=0.3,0.1

Type RM Length L Ch R = 1 ,7953    ,596,596,596
BEGIN DESCRIPTION:
Bitter Creek Trib14 9.0
END DESCRIPTION:
XS GIS Cut Line= 3
      1406554.96      6842588.01      1407860.68      6842390.31
      1408554.98        6842288.
#Sta/Elev= 30
  3679.4 2165.71  3708.8 2166.55  3782.6 2162.94  3978.6 2142.74  4023.3 2138.58
  4042.7 2134.55  4094.1 2135.51  4134.6 2130.32  4312.8 2121.69  4668.7 2118.94
    4704 2118.82  4894.8 2117.74  4963.9    2114  4985.6 2109.57  4987.5 2107.39
    4988 2106.89  5011.9 2107.39    5050 2114.77    5065 2112.87  5106.1 2112.67
  5206.5 2113.16    5254 2110.88  5307.6  2111.7  5407.6 2117.21  5499.7 2126.43
  5519.9 2125.91  5590.6  2131.9  5651.3 2137.96  5680.1 2143.48  5701.8 2151.96
#Mann= 10 ,-1 , 0
  3679.4     .07       0  3978.6    .035       0  4668.7     .07       0
    4704     .16       0  4894.8     .12       0  4987.5     .07       0
  5011.9     .12       0  5106.1     .12       0  5407.6    .035       0
  5680.1     .16       0
Bank Sta=4987.5,5011.9
XS Rating Curve= 0 ,0
Exp/Cntr=0.3,0.1

Type RM Length L Ch R = 1 ,7357    ,454,454,454
BEGIN DESCRIPTION:
Bitter Creek Trib14 8.0
END DESCRIPTION:
XS GIS Cut Line= 3
      1406604.98        6842688.      1407904.56      6842943.18
      1408605.02      6842387.99
#Sta/Elev= 30
  3675.6 2166.42  3866.9 2148.99  3899.8 2142.86  3930.4 2143.17  3981.4 2136.51
  4195.4  2123.4  4443.5 2119.42  4543.8 2117.56    4848 2115.67  4908.7 2113.67
  4929.1 2108.46  4980.1 2106.43  5058.5 2109.57  5177.3 2106.27  5177.8 2105.77
  5201.8 2106.27  5210.3 2108.25  5359.3 2109.88  5423.4 2106.31  5446.3 2110.46
  5452.3 2110.14  5466.7 2117.25    5502 2115.29  5523.7 2117.63  5545.3 2115.62
  5634.2  2117.9  5756.3 2125.31    5808 2131.13  5865.8 2148.63  5893.8 2153.24
#Mann= 10 ,-1 , 0
  3675.6     .07       0  3866.9    .035       0  4443.5     .07       0
  4543.8    .035       0  5058.5     .15       0  5177.3    .035       0
  5201.8     .15       0  5446.3     .16       0  5634.2    .035       0
  5756.3     .16       0
Bank Sta=5177.3,5201.8
XS Rating Curve= 0 ,0
Exp/Cntr=0.3,0.1

Type RM Length L Ch R = 1 ,6903    ,822,822,822
BEGIN DESCRIPTION:
Bitter Creek Trib14 7.0
END DESCRIPTION:
XS GIS Cut Line= 3
      1406940.92      6843256.96      1407804.12      6843322.64
      1408760.17      6842944.54
#Sta/Elev= 30
  4134.3 2130.96  4810.3 2117.51  4874.3 2115.21    4958  2106.9  4970.8  2106.4
  4985.7 2102.96  4986.2 2102.46  5010.2 2102.96  5021.6 2104.46    5027 2103.45
  5056.7 2107.25  5233.5  2109.9    5259 2110.98  5321.7  2109.7  5420.3 2115.41
  5435.3 2114.43    5465 2115.69    5673 2114.56    5711 2115.37  5759.7 2114.02
  5765.1 2117.72  5775.2 2116.74  5789.4 2117.74  5807.5 2116.59  5819.2 2114.31
  5866.4  2116.2  5946.3 2119.21    5976 2122.08  6005.8 2122.13  6028.1 2124.52
#Mann= 7 ,-1 , 0
  4134.3    .035       0    4958     .15       0  4985.7     .07       0
  5010.2     .15       0  5233.5     .16       0    5673     .07       0
  5866.4    .035       0
Bank Sta=4985.7,5010.2
XS Rating Curve= 0 ,0
Exp/Cntr=0.3,0.1

Type RM Length L Ch R = 1 ,6081    ,459,459,459
BEGIN DESCRIPTION:
Bitter Creek Trib14 6.0
END DESCRIPTION:
XS GIS Cut Line= 3
      1407513.82      6844062.53      1408138.73      6843720.69
      1408805.02      6842937.98
#Sta/Elev= 30
  4287.7 2126.02    4460 2120.44  4726.8 2108.22  4785.8 2105.65  4976.5 2102.51
    5006 2100.39    5008 2099.04  5008.5 2098.54  5032.6 2099.04  5035.4 2099.54
  5063.1 2102.84    5084 2107.12    5106 2107.82  5120.3 2110.74  5134.5 2111.64
  5239.8 2111.56  5390.1 2112.57  5491.2 2112.89  5701.2 2113.19  5737.4 2115.68
  5751.7 2113.99  5763.2 2115.16  5786.8  2114.5  5793.4 2116.66  5815.4 2115.48
  5879.1 2117.92  5914.2 2121.51  5942.8  2121.7  5992.2 2127.66  6027.9 2128.77
#Mann= 9 ,-1 , 0
  4287.7    .035       0  4726.8    .033       0    5008    .033       0
  5032.6    .033       0  5035.4     .15       0  5239.8     .07       0
  5390.1     .16       0  5491.2     .07       0  5763.2    .035       0
Bank Sta=5008,5032.6
XS Rating Curve= 0 ,0
Exp/Cntr=0.3,0.1

Type RM Length L Ch R = 1 ,5622    ,595,595,595
BEGIN DESCRIPTION:
Bitter Creek Trib14 5.0
END DESCRIPTION:
XS GIS Cut Line= 3
      1407905.01      6844437.99      1408218.56      6844151.24
        1409005.        6843338.
#Sta/Elev= 30
  4575.1 2131.99  4681.5 2133.66  4737.7 2130.43  4780.1  2125.5  4836.9 2124.01
  4852.8 2122.23  4879.9 2120.02  4900.4 2117.44  4907.8 2112.92  4928.7 2109.63
  4950.3 2101.05  4966.3 2097.48  4966.8 2096.98  4991.1 2097.48  5020.9 2100.69
  5056.4 2101.04  5063.4 2102.67  5077.5 2101.75  5136.7 2105.19  5170.2 2107.71
  5358.5 2108.79  5827.1 2111.29  5926.2 2113.15  6017.2 2117.95  6046.5 2119.99
  6060.7 2122.85  6098.9 2125.08  6124.2 2127.68  6127.8 2129.66  6131.3 2129.66
#Mann= 10 ,-1 , 0
  4575.1    .063       0  4852.8    .035       0  4879.9    .033       0
  4966.3    .033       0  4991.1    .033       0  5136.7     .15       0
  5170.2    .033       0  5358.5     .16       0  6017.2    .035       0
  6098.9    .063       0
Bank Sta=4966.3,4991.1
XS Rating Curve= 0 ,0
Exp/Cntr=0.3,0.1

Type RM Length L Ch R = 1 ,5027    ,550,550,550
BEGIN DESCRIPTION:
Bitter Creek Trib14 4.0
END DESCRIPTION:
XS GIS Cut Line= 3
      1408105.03      6845037.97      1408575.31      6844607.87
      1409305.01        6844338.
#Sta/Elev= 30
  4362.7 2147.18    4366 2147.18  4369.7 2143.68  4390.7 2140.79  4398.1 2131.76
  4404.9 2130.44  4412.3 2126.67  4419.1  2127.6  4454.9 2125.27  4504.2 2124.84
  4555.7 2120.91  4765.8 2109.45  4815.6 2106.49  4886.5 2099.62    4966 2095.58
  4966.5 2095.08  4990.9 2095.58  5020.9 2097.23  5127.6 2100.87    5217 2104.97
  5444.3 2106.22    5591 2108.54  5651.8 2112.31  5671.4 2114.38  5687.4 2118.18
    5702 2123.18    5714 2125.55  5737.7 2126.64  5756.7 2136.05    5778 2137.89
#Mann= 8 ,-1 , 0
  4362.7    .063       0  4555.7    .035       0  4765.8    .033       0
    4966    .033       0  4990.9    .033       0  5020.9     .12       0
  5127.6    .033       0  5687.4    .063       0
Bank Sta=4966,4990.9
XS Rating Curve= 0 ,0
Exp/Cntr=0.3,0.1

Type RM Length L Ch R = 1 ,4477    ,597,597,597
BEGIN DESCRIPTION:
Bitter Creek Trib14 3.0
END DESCRIPTION:
XS GIS Cut Line= 3
      1408455.03      6845337.97      1408798.89      6845085.82
      1409505.03      6844687.98
#Sta/Elev= 30
  4573.6 2140.62  4623.2 2139.81  4645.7 2133.96  4651.9 2130.19  4660.4  2129.1
  4687.4 2120.88  4702.1 2119.09  4716.7  2119.7  4722.9 2117.27  4731.4 2117.91
  4737.6 2114.89  4786.7 2107.64  4842.2 2099.58  4881.9 2096.09  4991.1 2093.36
  4991.6 2092.86    5016 2093.36  5161.3 2102.22    5489 2106.19  5626.8 2113.52
  5649.8 2115.33  5669.7 2119.87  5684.2 2123.92  5699.9 2124.31  5707.2 2128.72
  5715.8 2130.09  5737.5 2130.36  5759.2 2134.17  5785.2 2134.28  5810.5 2135.67
#Mann= 8 ,-1 , 0
  4573.6    .035       0  4786.7    .033       0  4842.2     .12       0
  4991.1     .07       0    5016     .12       0  5161.3    .033       0
  5669.7    .063       0  5785.2    .035       0
Bank Sta=4991.1,5016
XS Rating Curve= 0 ,0
Exp/Cntr=0.3,0.1
