--- Bluff Creek.prj (project) ---

Proj Title=Bluff Creek Base Level Engineering
Current Plan=p01
Default Exp/Contr=0.3,0.1
English Units
Geom File=g01
Flow File=f01
Plan File=p01
Y Axis Title=Elevation
X Axis Title(PF)=Main Channel Distance
X Axis Title(XS)=Station
BEGIN DESCRIPTION:
Bluff Creek
END DESCRIPTION:
DSS Export Rating Curves= 0
DSS Export Rating Curve Sorted= 0
DSS Export Volume Flow Curves= 0
DXF OffsetX= 0
DXF OffsetY= 0
DXF ScaleX= 1
DXF ScaleY= 10

--- Bluff Creek.p01 (plan) ---

Plan Title=Multiple Run
Short Identifier=Multiple
Geom File=g01
Flow File=f01
Subcritical Flow
K Sum by GR= 0
Std Step Tol= 0.01
Critical Tol= 0.01
Num of Std Step Trials= 20
Max Error Tol= 0.3
Flow Tol Ratio= 0.001
Split Flow NTrial= 30
Split Flow Tol= 0.02
Split Flow Ratio= 0.02
Log Output Level= 0
Friction Slope Method= 1
Unsteady Friction Slope Method= 2
Unsteady Bridges Friction Slope Method= 1
Parabolic Critical Depth
Global Vel Dist=  1 , 1 , 1
Global Log Level= 0
CheckData=True
Encroach Param= -1, 0, 0, 0
BEGIN DESCRIPTION:
Multiple Run
END DESCRIPTION:

--- Bluff Creek.f01 (steady flow) ---

Flow Title=Multiple
Number of Profiles=7
Profile Names=10-year,25-year,50-year,1pct_min,100-year,1pct_plu,500-year
River Rch & RM= Bluff Creek,Reach-1,23576
     317     448     559     347     692    1380    1072
River Rch & RM= Bluff Creek,Reach-1,19683
     859    1287    1666    1070    2134    4258    3549
River Rch & RM= Bluff Creek,Reach-1,15752
    1185    1785    2320    1492    2977    5941    4972
River Rch & RM= Bluff Creek,Reach-1,13758
    1271    1920    2499    1610    3212    6409    5380
River Rch & RM= Bluff Creek,Reach-1,10910
    1296    1959    2550    1643    3279    6542    5494
River Rch & RM= Bluff Creek,Reach-1,10311
    1360    2055    2676    1724    3441    6865    5765
River Rch & RM= Bluff Creek,Reach-1,8597
    1318    1982    2572    1651    3294    6572    5477
Boundary for River Rch & Prof#=Bluff Creek,Reach-1,1
Up Type=0
Dn Type=3
Dn Slope=0.005
Boundary for River Rch & Prof#=Bluff Creek,Reach-1,2
Up Type=0
Dn Type=3
Dn Slope=0.005
Boundary for River Rch & Prof#=Bluff Creek,Reach-1,3
Up Type=0
Dn Type=3
Dn Slope=0.005
Boundary for River Rch & Prof#=Bluff Creek,Reach-1,4
Up Type=0
Dn Type=3
Dn Slope=0.005
Boundary for River Rch & Prof#=Bluff Creek,Reach-1,5
Up Type=0
Dn Type=3
Dn Slope=0.005
Boundary for River Rch & Prof#=Bluff Creek,Reach-1,6
Up Type=0
Dn Type=3
Dn Slope=0.005
Boundary for River Rch & Prof#=Bluff Creek,Reach-1,7
Up Type=0
Dn Type=3
Dn Slope=0.005

--- Bluff Creek.g01 (geometry) ---

Geom Title=Existing Conditions
Program Version=4.10

River Reach=Bluff Creek     ,Reach-1
Reach XY= 30
        1400855.        6887788.      1401232.32      6888088.11
      1401665.48      6887538.93      1402286.64      6887738.45
      1402402.29      6887443.28      1402839.93      6887438.18
      1403249.48      6887685.65      1404048.59      6886645.63
      1404499.45      6886833.23      1404312.34      6886231.67
      1404988.36      6886204.75      1405068.47      6885674.43
      1406149.53      6884790.45      1406057.15      6884243.97
      1406512.81      6883431.81      1407149.67      6882990.66
      1406915.76      6882178.32      1407638.72      6881705.14
      1408349.54      6880890.45      1408510.18      6880093.41
      1409249.59      6879732.82      1409410.03      6879143.08
       1409797.2      6878994.21      1409831.27      6878211.11
       1410847.2      6878094.21      1410408.82      6877139.58
      1411149.83      6877032.59      1411108.54      6876389.44
      1411732.46      6876111.83        1411655.        6875838.

Type RM Length L Ch R = 1 ,23576   ,966,966,966
BEGIN DESCRIPTION:
Bluff Creek 37.0
END DESCRIPTION:
XS GIS Cut Line= 3
        1401305.      6888338.05      1401325.28      6888038.53
      1401055.01      6887288.02
#Sta/Elev= 30
  4699.8 2061.44  4729.9 2059.89  4750.9 2056.73    4760 2055.15  4774.4 2056.76
  4800.1 2054.35  4820.1 2055.23  4850.2 2052.02  4870.2 2052.39  4910.3 2050.74
  4923.6 2049.78  4930.4 2047.88  4940.4  2046.8  4960.4 2045.73  4970.5 2042.68
  4978.3 2041.63  4978.6 2041.13  4982.7 2041.63  4997.8 2044.75    5016 2045.72
  5102.8 2046.42  5164.2 2048.59  5225.6 2048.99  5266.3 2047.73  5287.5 2049.85
  5382.6 2052.09  5581.1 2060.45  5664.9 2064.71  5776.5 2067.44  5797.7 2069.23
#Mann= 6 ,-1 , 0
  4699.8    .035       0  4750.9     .07       0  4978.3     .07       0
  4982.7     .07       0  5382.6     .16       0  5581.1     .07       0
Bank Sta=4978.3,4982.7
XS Rating Curve= 0 ,0
Exp/Cntr=0.3,0.1

Type RM Length L Ch R = 1 ,22610   ,499,499,499
BEGIN DESCRIPTION:
Bluff Creek 36.0
END DESCRIPTION:
XS GIS Cut Line= 3
      1401454.99      6888338.02      1401948.94      6887546.15
        1401955.      6887137.99
#Sta/Elev= 30
  4066.7 2060.53  4089.7 2057.59  4103.3 2057.39  4116.9 2058.49  4125.6 2056.79
  4153.4 2054.76  4174.7 2054.91  4226.6 2052.41  4290.7 2051.24  4314.2 2051.89
  4349.6  2049.8  4442.6 2048.27  4479.2 2048.71  4515.6 2046.98  4639.2 2045.47
  4661.9  2046.2  4704.4 2044.56  4735.1 2045.35  4893.1 2040.75  4929.7 2040.96
  4977.8 2039.65  4985.3 2039.41  4985.6 2038.91  4989.8 2039.41  5067.2 2043.72
  5072.2 2042.74  5136.5 2045.41  5357.1  2058.8  5398.2 2060.73  5408.2 2062.54
#Mann= 9 ,-1 , 0
  4066.7     .07       0  4103.3    .035       0  4442.6     .07       0
  4639.2    .035       0  4977.8     .07       0  4985.3     .07       0
  4989.8     .07       0  5136.5     .16       0  5357.1    .035       0
Bank Sta=4985.3,4989.8
XS Rating Curve= 0 ,0
Exp/Cntr=0.3,0.1

Type RM Length L Ch R = 1 ,22111   ,498,498,498
BEGIN DESCRIPTION:
Bluff Creek 35.0
END DESCRIPTION:
XS GIS Cut Line= 3
      1401854.99      6888538.02      1402311.36      6887730.68
        1402055.      6886987.99
#Sta/Elev= 30
  4072.6 2065.87  4183.1 2058.59  4204.4  2058.9  4242.3  2055.6  4341.5 2051.68
  4394.3 2048.55  4440.2 2048.79  4497.7 2046.19  4782.5 2043.32  4847.8 2043.07
  4938.1 2042.08  5003.4  2036.7  5011.2 2036.12  5011.5 2035.62  5015.7 2036.12
  5037.3 2037.97  5140.4 2038.79  5156.8 2037.62  5162.1 2038.94  5182.7 2037.58
  5250.4  2042.8  5267.3 2041.57  5304.8  2042.8  5410.2 2046.97  5552.3 2054.75
  5574.1 2053.43  5588.2 2055.22  5595.3 2057.62  5655.2 2061.06  5785.7 2070.46
#Mann= 12 ,-1 , 0
  4072.6    .045       0  4204.4    .035       0  4341.5     .07       0
  4782.5    .035       0  4847.8     .07       0  5003.4    .035       0
  5011.2     .07       0  5015.7    .035       0  5304.8     .07       0
  5410.2     .16       0  5552.3    .035       0  5655.2     .07       0
Bank Sta=5011.2,5015.7
XS Rating Curve= 0 ,0
Exp/Cntr=0.3,0.1

Type RM Length L Ch R = 1 ,21613   ,495,495,495
BEGIN DESCRIPTION:
Bluff Creek 34.0
END DESCRIPTION:
XS GIS Cut Line= 3
      1402255.01      6888587.97      1402560.53      6887485.63
      1402254.97      6887087.97
#Sta/Elev= 30
  3856.1 2050.35  3873.2 2051.32  4121.5 2045.54  4173.4    2046  4260.8  2042.9
  4286.7 2044.37  4302.3 2042.47  4871.3 2039.36  4959.9 2035.35  4976.8 2032.47
  5009.6 2032.41  5014.3 2030.26  5014.7 2029.76  5018.9 2030.26  5037.4 2030.99
  5045.6 2033.36  5051.7 2031.01  5060.1 2033.57  5066.4 2038.25  5072.1 2036.69
    5081 2038.69  5087.3  2036.6  5095.5 2038.05  5116.3 2036.87  5130.8  2040.7
  5184.3 2040.76  5228.8 2043.97  5316.3 2047.31  5422.6 2052.94  5501.5 2058.15
#Mann= 12 ,-1 , 0
  3856.1    .035       0  4121.5     .07       0  4871.3    .035       0
  4959.9     .07       0  5014.3     .07       0  5018.9     .07       0
  5051.7    .035       0  5072.1     .07       0  5184.3    .035       0
  5228.8     .16       0  5316.3    .035       0  5422.6     .07       0
Bank Sta=5014.3,5018.9
XS Rating Curve= 0 ,0
Exp/Cntr=0.3,0.1

Type RM Length L Ch R = 1 ,21118   ,438,438,438
BEGIN DESCRIPTION:
Bluff Creek 33.0
END DESCRIPTION:
XS GIS Cut Line= 3
       1402751.3      6887610.22      1402966.01      6887603.34
      1402993.44      6887513.03
#Sta/Elev= 30
  4846.4 2035.35  4880.1 2034.19  4900.1 2035.07  4910.1 2034.23  4920.1 2033.97
  4930.1 2032.78  4940.1 2030.25  4950.2 2029.56  4960.2 2027.62  4964.5 2026.39
  4970.2 2024.77  4980.2 2024.75  4987.9 2022.43  4988.2 2021.93  4992.2 2021.93
  4992.5 2022.43  5000.2 2023.99  5010.2 2031.12  5020.2 2032.69  5030.2 2034.06
  5040.2 2034.54  5073.5 2035.39  5078.4 2035.21  5087.7  2035.4  5098.2 2036.25
  5106.4 2037.46  5111.6  2036.9  5139.3 2038.37  5150.4 2038.51  5155.6  2039.3
#Mann= 5 ,-1 , 0
  4846.4     .07       0  4964.5     .16       0  4987.9     .07       0
  4992.5     .16       0  5078.4     .07       0
Bank Sta=4987.9,4992.5
XS Rating Curve= 0 ,0
Exp/Cntr=0.3,0.1

Type RM Length L Ch R = 1 ,20680   ,236,236,236
BEGIN DESCRIPTION:
Bluff Creek 32.0
END DESCRIPTION:
XS GIS Cut Line= 3
        1403255.      6887787.97      1403241.09      6887687.33
      1403004.98      6887437.98
#Sta/Elev= 30
  4898.4 2039.63  4918.6 2037.58  4934.3 2036.99  4939.3  2038.3  4948.8 2036.65
  4958.9 2034.19    4969 2032.94  4979.1 2030.39  4989.2 2026.49  4997.1 2023.99
  5003.8 2023.36    5011 2020.39  5022.9 2019.38  5023.2 2018.88  5027.2 2018.88
  5027.6 2019.38  5039.4 2022.31  5046.2 2023.19  5053.5 2026.03  5060.4 2027.17
  5067.7 2030.55  5074.6 2030.22  5081.7 2032.44  5095.6 2033.39  5106.1 2033.55
  5138.1 2034.06  5145.4    2035  5159.8 2035.55  5237.2 2036.83  5343.4  2039.8
#Mann= 5 ,-1 , 0
  4898.4     .07       0  5022.9     .07       0  5027.6     .07       0
  5106.1     .16       0  5159.8     .07       0
Bank Sta=5022.9,5027.6
XS Rating Curve= 0 ,0
Exp/Cntr=0.3,0.1

Type RM Length L Ch R = 1 ,20444   ,263,263,263
BEGIN DESCRIPTION:
Bluff Creek 4447
END DESCRIPTION:
XS GIS Cut Line= 3
      1403512.97      6887709.59      1403444.97       6887587.9
      1403158.73      6887454.97
#Sta/Elev= 30
  4860.6 2040.73  4863.6 2040.73  4873.9 2038.83  4889.1  2038.6  4910.8 2036.49
  4919.7 2034.57  4926.8 2031.22  4932.5 2032.18  4942.6 2027.56  4948.5 2023.03
  4964.5 2014.85  4974.6 2013.48  4974.9 2012.98    4979 2012.98  4979.4 2013.48
  4991.9 2014.87 5015.35 2021.61 5027.52 2023.05 5027.52 2024.27  5031.5 2024.93
    5037 2028.08  5044.1 2028.37  5059.9  2030.9  5082.8  2031.4  5088.3 2032.61
  5165.4 2034.02  5197.2 2034.03  5264.6 2035.59  5271.4  2036.3  5315.6 2036.63
#Mann= 3 ,-1 , 0
  4860.6     .07       0  4974.6     .07       0  4979.4     .07       0
Bank Sta=4974.6,4979.4
XS Rating Curve= 0 ,0
Exp/Cntr=0.3,0.1

Type RM Length L Ch R = 1 ,20181   ,498,498,498
BEGIN DESCRIPTION:
Bluff Creek 31.0
END DESCRIPTION:
XS GIS Cut Line= 3
      1403712.41      6887546.47      1403554.33      6887401.93
      1403264.13      6887323.15
#Sta/Elev= 30
  4785.8 2040.38  4846.7 2038.32  4896.1  2033.4  4924.4 2032.04  4938.6 2030.38
  4945.4 2029.28  4952.8 2025.33  4959.6 2018.03    4967 2013.61  4971.4 2013.38
  4971.7 2012.88  4976.2 2013.38  4995.4 2014.93  5002.2 2014.27    5020 2017.67
  5029.6 2022.05  5034.8 2019.74  5040.8 2022.65  5061.5 2024.76  5069.5 2027.14
  5074.6 2023.45  5092.6 2025.03  5109.3 2028.41  5123.7 2027.65  5143.9 2028.34
  5149.1 2026.52  5165.1 2027.16  5228.7 2033.92  5294.1 2037.36  5300.7 2037.27
#Mann= 4 ,-1 , 0
  4785.8     .07       0  4971.4     .07       0  4976.2     .07       0
  5294.1     .16       0
Bank Sta=4971.4,4976.2
XS Rating Curve= 0 ,0
Exp/Cntr=0.3,0.1

Type RM Length L Ch R = 1 ,19683   ,491,491,491
BEGIN DESCRIPTION:
Bluff Creek 30.0
END DESCRIPTION:
XS GIS Cut Line= 3
      1403709.51        6887253.      1403693.18      6887050.46
      1403555.03      6886988.01
#Sta/Elev= 30
  4796.8 2031.27  4811.8 2030.14    4862 2029.14  4902.1 2025.73  4911.1 2023.65
  4916.1 2025.02  4922.2 2024.16  4942.3 2023.39  4962.3 2021.27  4972.4 2018.87
  4982.4 2007.45    4987 2003.74  4987.5 2003.24  4997.3 2003.24  4997.8 2003.74
  4998.7 2005.28    5009 2008.06  5021.8 2012.94  5044.9 2014.87    5068 2015.09
  5085.6 2018.84  5091.1 2024.76  5096.8  2027.1  5107.7 2026.99  5114.2 2032.61
  5119.7 2032.27  5137.3 2039.35  5142.8  2039.2  5148.9 2041.15  5151.6 2041.15
#Mann= 3 ,-1 , 0
  4796.8     .07       0    4987     .07       0  4997.8     .07       0
Bank Sta=4987,4997.8
XS Rating Curve= 0 ,0
Exp/Cntr=0.3,0.1

Type RM Length L Ch R = 1 ,19192   ,497,497,497
BEGIN DESCRIPTION:
Bluff Creek 29.0
END DESCRIPTION:
XS GIS Cut Line= 4
      1404013.22      6887052.43        1404005.        6886838.
      1404001.11      6886736.56      1403808.98      6886609.95
#Sta/Elev= 30
  4683.9 2035.41  4722.3 2034.64  4748.4  2031.1  4778.4 2029.12  4920.8 2024.45
  4938.5 2022.42  4948.5 2018.93  4958.5 2014.26  4978.5 2011.09  4996.8 2001.14
  4998.5 2001.06    4999 2000.56  5009.4 2001.06  5009.9 2003.32    5019 2007.67
    5025 2009.31  5112.3 2016.53  5127.1 2018.92  5139.4 2022.17  5148.5 2022.42
  5154.4 2024.63  5169.5  2026.2  5175.5 2025.67  5184.6 2026.79  5190.6 2026.03
  5198.9 2027.87  5205.7 2031.66  5211.6 2032.02  5226.7 2037.64  5230.1 2035.84
#Mann= 5 ,-1 , 0
  4683.9     .07       0  4722.3     .16       0  4920.8     .07       0
  4998.5     .07       0  5009.4     .07       0
Bank Sta=4998.5,5009.4
XS Rating Curve= 0 ,0
Exp/Cntr=0.3,0.1

Type RM Length L Ch R = 1 ,18695   ,170,170,170
BEGIN DESCRIPTION:
Bluff Creek 28.0
END DESCRIPTION:
XS GIS Cut Line= 4
      1404222.05      6887093.21        1404305.        6886888.
      1404348.68      6886779.93        1404305.        6886638.
#Sta/Elev= 30
  4662.1 2041.47  4683.6 2040.41  4700.1 2036.13  4731.9 2037.75  4743.2  2034.4
    4754 2033.52  4766.8 2035.14    4795 2030.45  4834.9 2023.35  4915.8 2019.46
  4937.4 2011.88  4969.7 2009.44    4976 2001.53  4985.8 1999.45  4986.3 1998.95
  4996.7 1999.45  4998.3 2001.43  5012.5 2001.97  5028.8 2007.21  5034.1 2002.86
  5043.9 2004.93  5054.3 2009.91  5061.5 2010.73  5066.8 2008.84  5075.3 2013.57
  5094.2 2018.45  5099.5 2014.51  5106.7 2020.01  5135.3  2021.7  5148.5 2021.98
#Mann= 6 ,-1 , 0
  4662.1     .07       0    4795     .16       0  4834.9     .07       0
  4985.8     .07       0  4996.7     .07       0  5135.3     .16       0
Bank Sta=4985.8,4996.7
XS Rating Curve= 0 ,0
Exp/Cntr=0.3,0.1

Type RM Length L Ch R = 1 ,18525   ,328,328,328
BEGIN DESCRIPTION:
Bluff Creek 27.1
END DESCRIPTION:
XS GIS Cut Line= 3
      1404581.94        6887103.      1404499.45      6886833.23
      1404334.25      6886612.13
#Sta/Elev= 30
  4717.9 2038.45  4726.6 2037.74    4754 2038.67  4900.9 2031.62  4911.4 2028.83
  4921.8 2022.35  4933.6 2012.55  4953.2 2010.18  4984.6 2010.22  4999.1 2000.27
  5006.5 1997.53  5014.3  1997.6  5028.9 2001.71  5035.1 2001.15  5043.5 2004.21
  5049.7 1998.65  5064.3 2003.17  5065.1 1997.26  5065.6 1996.76    5076 1997.26
  5078.9 2000.14  5085.1 1997.29  5099.7 1997.96  5114.3 2002.45  5120.6 2002.23
  5135.2 2009.02  5143.5 2014.84  5156.3 2019.06  5263.4 2020.87    5276 2021.29
#Mann= 5 ,-1 , 0
  4717.9     .16       0  4726.6     .07       0  5065.1     .07       0
    5076     .07       0  5263.4     .16       0
Bank Sta=5065.1,5076
XS Rating Curve= 0 ,0
Exp/Cntr=0.3,0.1

Type RM Length L Ch R = 1 ,18197   ,473,473,473
BEGIN DESCRIPTION:
Bluff Creek 27.0
END DESCRIPTION:
XS GIS Cut Line= 4
      1404725.78      6886773.21        1404605.        6886588.
      1404505.47      6886533.26      1404355.02      6886587.99
#Sta/Elev= 30
  4665.3 2042.15  4670.7 2040.85  4712.9 2038.63  4719.3 2037.42  4821.5 2032.95
  4827.5 2031.67  4889.3 2026.72  4900.2 2022.93  4909.2 2021.32  4914.8 2017.65
  4921.9 2013.81    4938 2008.59  4954.1  2008.7  4959.8 2009.55  4975.9 2005.79
  4981.6 2006.33  4997.4 1999.33  5002.9 1999.33  5005.7 1996.68  5006.2 1996.18
  5016.6 1996.68  5021.8 2001.47  5027.8 2005.45    5075 2007.36  5096.3 2009.75
  5106.9 2009.99  5114.2 2013.72  5119.6 2013.93  5128.2 2018.13  5160.1 2020.25
#Mann= 4 ,-1 , 0
  4665.3     .07       0  4914.8     .16       0  5005.7     .07       0
  5016.6     .16       0
Bank Sta=5005.7,5016.6
XS Rating Curve= 0 ,0
Exp/Cntr=0.3,0.1

Type RM Length L Ch R = 1 ,17724   ,587,587,587
BEGIN DESCRIPTION:
Bluff Creek 26.0
END DESCRIPTION:
XS GIS Cut Line= 3
      1404707.39      6886474.84      1404386.46       6886187.3
      1404008.22      6886140.75
#Sta/Elev= 30
  4569.1 2028.11  4589.6 2025.55  4649.4 2023.57  4800.8  2020.1  4813.1 2020.13
  4866.3 2017.31  4904.1 2011.07    4944 2005.64  4986.6 2003.05  4993.4 2000.01
  5011.5 2000.14  5029.9 1996.65  5030.4 1996.15  5042.1 1996.65  5061.9 1998.19
  5082.1 2006.36  5092.2 2007.15  5117.2 2000.14  5142.5 2003.47  5198.4 2002.18
  5203.5 2004.27  5213.1 2001.56  5243.3 2010.61  5253.4 2015.72  5279.7 2018.76
  5284.7 2016.23  5303.7    2018  5323.9 2023.87  5349.7 2026.44  5381.1    2032
#Mann= 8 ,-1 , 0
  4569.1     .07       0  4649.4     .16       0  4800.8     .07       0
  4813.1     .16       0  4904.1     .07       0  5029.9     .07       0
  5042.1     .07       0  5349.7    .035       0
#XS Ineff= 2 , 0
                         5087.31         2013.77
Permanent Ineff=
       F       F
Bank Sta=5029.9,5042.1
XS Rating Curve= 0 ,0
Exp/Cntr=0.3,0.1

Type RM Length L Ch R = 1 ,17137   ,402,402,402
BEGIN DESCRIPTION:
Bluff Creek 25.0
END DESCRIPTION:
XS GIS Cut Line= 3
      1404971.68      6886366.33      1404911.75       6886278.9
      1404503.56      6885886.22
#Sta/Elev= 30
    4894 2045.87  4933.4 2041.63  4948.3 2020.25  4963.2 2007.75  4976.8 1998.33
  4991.4  1994.3  4991.9  1993.8  5003.6  1994.3  5026.6 2000.74  5062.1 2001.26
    5069 2005.98  5076.2 2003.26  5093.7  2004.8  5132.8 2005.16  5153.9 2009.43
  5161.1 2006.32  5179.3 2008.14  5186.3 2009.16  5210.5 2011.95  5217.5 2016.92
  5224.7  2026.4  5238.8  2031.1    5274 2033.64  5281.3 2036.78  5359.3 2034.21
  5401.4 2025.84    5458 2022.11  5500.4  2022.8    5536 2035.46  5566.4 2031.44
#Mann= 7 ,-1 , 0
    4894     .07       0  4991.4     .07       0  5003.6     .07       0
  5093.7     .16       0  5179.3     .07       0  5186.3     .16       0
  5359.3     .07       0
Bank Sta=4991.4,5003.6
XS Rating Curve= 0 ,0
Exp/Cntr=0.3,0.1

Type RM Length L Ch R = 1 ,16735   ,496,496,496
BEGIN DESCRIPTION:
Bluff Creek 24.0
END DESCRIPTION:
XS GIS Cut Line= 3
      1405180.82       6885961.7      1405013.14      6885944.06
      1404905.01        6885938.
#Sta/Elev= 30
  4831.4 2019.84  4837.1 2019.47  4877.5 2014.96  4887.5 2014.69  4897.6 2013.58
  4907.6 2008.63  4913.6 2006.54  4918.6 2006.29  4927.7 2004.73  4957.9 2001.51
    4968 1999.72    4978 1995.72  4988.1 1993.81  4990.5 1992.28    4991 1991.78
  5002.2 1991.78  5002.7 1992.28  5008.2 1994.73    5016 1996.65    5021 1995.26
  5026.4 1999.98  5028.2 2001.55  5038.2 2004.72  5048.2 2005.57  5058.2 2008.41
  5068.2 2009.89  5088.3 2014.19  5098.3 2014.74  5105.8 2015.94  5108.3 2015.94
#Mann= 5 ,-1 , 0
  4831.4     .07       0  4837.1     .16       0  4990.5     .07       0
  5002.7     .16       0  5026.4     .07       0
Bank Sta=4990.5,5002.7
XS Rating Curve= 0 ,0
Exp/Cntr=0.3,0.1

Type RM Length L Ch R = 1 ,16239   ,487,487,487
BEGIN DESCRIPTION:
Bluff Creek 23.0
END DESCRIPTION:
XS GIS Cut Line= 3
      1405254.99      6885687.96      1405231.69      6885561.39
      1405155.03      6885488.03
#Sta/Elev= 30
  4871.3 2011.11  4873.8 2011.11  4881.4    2009  4891.6 2007.53  4897.8 2006.14
  4902.9  2006.8  4905.2 2006.08  4911.9 2003.99  4922.1 2002.91  4932.3 2003.15
  4944.1 2000.99  4955.9 2000.41  4962.8 1997.53  4972.9 1993.91  4983.1 1991.84
  4987.1 1990.41  4987.6 1989.91  4998.9 1989.91  4999.4 1990.41  5014.2 2000.89
  5021.4 2004.94  5035.5 2014.52  5042.5 2024.31  5049.7 2031.41  5056.6 2033.58
  5070.8 2033.59  5084.9 2032.51  5092.2 2032.66  5099.1  2031.7  5106.1 2031.88
#Mann= 5 ,-1 , 0
  4871.3     .07       0  4905.2     .16       0  4944.1     .07       0
  4987.1     .07       0  4999.4     .07       0
Bank Sta=4987.1,4999.4
XS Rating Curve= 0 ,0
Exp/Cntr=0.3,0.1

Type RM Length L Ch R = 1 ,15752   ,496,496,496
BEGIN DESCRIPTION:
Bluff Creek 22.0
END DESCRIPTION:
XS GIS Cut Line= 3
        1405655.      6885487.98      1405611.07      6885279.87
      1405404.98        6885238.
#Sta/Elev= 30
  4787.3 2016.02  4807.1 2014.78  4817.9 2012.81  4838.4 2013.63  4899.7 2010.73
  4911.7 2007.66  4920.1 2007.69  4940.6 2001.66  4950.8  1995.8  4982.5 1990.82
    4983 1990.32  5000.9 1990.82  5006.2 1991.31  5026.6 1996.83  5033.1 1997.39
  5038.2 2000.21  5077.6 1999.98  5088.8 2001.57  5108.2 2008.26  5122.1 2010.39
  5128.6 2010.29  5131.2 2011.54  5134.3 2013.02  5159.3  2017.9  5169.5 2018.75
  5179.7 2023.45    5185 2028.76  5190.1  2032.3  5200.1 2035.16  5210.3 2035.34
#Mann= 5 ,-1 , 0
  4787.3     .07       0  4982.5     .07       0  5000.9     .07       0
  5122.1     .16       0  5131.2     .07       0
Bank Sta=4982.5,5000.9
XS Rating Curve= 0 ,0
Exp/Cntr=0.3,0.1

Type RM Length L Ch R = 1 ,15256   ,383,383,383
BEGIN DESCRIPTION:
Bluff Creek 21.0
END DESCRIPTION:
XS GIS Cut Line= 3
      1406154.98      6885087.99      1405975.27      6884988.52
      1405754.99        6884938.
#Sta/Elev= 30
  4794.6 2022.99  4817.4 2020.04  4840.3 2020.16  4851.8 2017.04  4862.1 2020.13
  4867.9 2016.74  4883.9  2024.1  4889.6 2017.88  4905.7 2014.39  4927.4 2006.25
  4933.1 2002.32  4949.2 1998.53  4970.9 1997.22    4987 1991.98    4988 1986.18
  4988.5 1985.68  5006.5 1986.18  5010.5  1987.2  5020.2 1987.94  5025.3 1991.68
  5051.6 1992.72  5061.8 1996.27  5068.2 2000.41  5073.3 2005.78  5082.4 2004.55
  5092.6 2006.56  5111.1 2006.68  5116.2 2008.77  5133.7 2010.71    5226 2013.09
#Mann= 3 ,-1 , 0
  4794.6     .07       0    4988     .07       0  5006.5     .07       0
Bank Sta=4988,5006.5
XS Rating Curve= 0 ,0
Exp/Cntr=0.3,0.1

Type RM Length L Ch R = 1 ,14873   ,234,234,234
BEGIN DESCRIPTION:
Bluff Creek 20.1
END DESCRIPTION:
XS GIS Cut Line= 3
      1406438.84      6884755.92      1406155.16        6884688.
      1405679.43      6884626.37
#Sta/Elev= 30
  4708.3 2030.12  4719.1  2029.4  4724.3 2025.69  4732.8 2025.13  4815.1 2024.64
  4825.4 2023.06  4850.4 2022.49  4917.9 2021.89  4934.5 2025.71  4939.6 2022.61
    4959 2021.96  4969.3 2016.98  4976.5 1996.66    5000 1989.49    5001 1985.79
  5001.5 1985.29  5019.5 1985.79  5020.3 1991.77  5037.2 1997.29  5090.9 1997.27
  5111.1 2000.45  5195.7 2002.99  5242.2 2006.42  5269.2 2009.82  5363.2 2014.84
  5403.5 2018.68  5423.4 2018.11  5443.8 2022.54    5464 2025.04  5479.7 2022.75
#Mann= 4 ,-1 , 0
  4708.3     .07       0    5001     .07       0  5019.5     .07       0
  5269.2    .035       0
Bank Sta=5001,5019.5
XS Rating Curve= 0 ,0
Exp/Cntr=0.3,0.1

Type RM Length L Ch R = 1 ,14639   ,382,382,382
BEGIN DESCRIPTION:
Bluff Creek 20.0
END DESCRIPTION:
XS GIS Cut Line= 3
      1406402.92      6884523.53      1406060.13      6884490.28
      1405755.04        6884488.
#Sta/Elev= 30
  4655.6 2022.86  4659.8  2021.8  4683.7 2020.34  4703.7 2017.31  4743.9  2017.5
  4761.8 2019.55  4804.2 2020.13  4834.4 2015.64  4863.9 2014.04  4874.5 2011.58
  4894.6 2010.46  4904.7 2006.29  4914.7 1999.28  4924.8 1996.69  4944.9  1993.9
  4954.9 1990.26  4955.7 1985.65  4956.2 1985.15  4974.2 1985.65    4995 1995.01
    5000 1995.01  5005.1 1998.19  5065.1 2001.69  5125.1 2008.97  5191.9 2014.64
  5225.1 2019.06  5245.1 2020.53  5265.1 2024.45  5285.1 2026.18  5305.1 2031.28
#Mann= 4 ,-1 , 0
  4655.6     .07       0  4955.7     .07       0  4974.2     .07       0
  5191.9    .035       0
Bank Sta=4955.7,4974.2
XS Rating Curve= 0 ,0
Exp/Cntr=0.3,0.1

Type RM Length L Ch R = 1 ,14257   ,499,499,499
BEGIN DESCRIPTION:
Bluff Creek 19.0
END DESCRIPTION:
XS GIS Cut Line= 3
      1406455.04      6884288.01      1406105.81      6884153.33
      1405904.99      6884288.01
#Sta/Elev= 30
  4625.7 2017.42  4665.3 2018.47  4679.3 2014.02  4700.8 2010.89  4711.5 2007.29
  4732.9 2008.96  4755.3 2004.21  4779.9 2003.58  4812.1 2005.33    4881 2000.78
  4894.4 1997.42    4958 1995.47  4979.4 1996.43  5003.5 1994.39  5012.2 1990.41
  5015.7 1985.49  5016.2 1984.99  5034.4 1985.49  5048.2 1990.51  5054.2 1989.81
  5064.3 1995.32  5101.8 2009.65  5120.2 2011.96  5126.2 2009.31  5141.2 2013.67
  5183.3 2020.48  5213.3 2022.63  5228.3 2024.36  5234.3 2027.06  5241.8 2027.15
#Mann= 7 ,-1 , 0
  4625.7     .07       0  4812.1     .16       0    4881     .07       0
  5015.7     .07       0  5034.4     .07       0  5064.3     .16       0
  5101.8     .07       0
Bank Sta=5015.7,5034.4
XS Rating Curve= 0 ,0
Exp/Cntr=0.3,0.1

Type RM Length L Ch R = 1 ,13758   ,496,496,496
BEGIN DESCRIPTION:
Bluff Creek 18.0
END DESCRIPTION:
XS GIS Cut Line= 3
      1406805.02      6884038.01       1406407.7      6883794.12
      1406204.99        6883788.
#Sta/Elev= 30
  4533.8  2025.2  4547.4  2024.2  4578.2 2018.04  4605.4 2013.93  4636.3 2011.75
  4721.6 2008.06  4830.3 2005.97  4862.4 2004.69  4889.6 2002.31  4897.6 1998.23
    4905  1990.8  4910.9 1990.53  4920.4 1986.48  4926.3 1986.31  4941.7 1994.47
  4956.2 1994.34  4968.9 1991.23  4974.5 1983.93    4975 1983.43    4994 1983.93
  4998.7 1990.52  5003.9 1990.52  5022.7 1995.78  5037.4 1995.91  5082.7 1999.63
  5101.1 2003.52  5112.8  2005.6  5152.8 2019.01  5162.8 2020.17  5202.8 2019.38
#Mann= 5 ,-1 , 0
  4533.8     .07       0  4830.3     .16       0  4974.5     .07       0
    4994     .16       0  5101.1     .07       0
Bank Sta=4974.5,4994
XS Rating Curve= 0 ,0
Exp/Cntr=0.3,0.1

Type RM Length L Ch R = 1 ,13262   ,492,492,492
BEGIN DESCRIPTION:
Bluff Creek 17.0
END DESCRIPTION:
XS GIS Cut Line= 3
      1407004.96      6883437.99      1406571.57      6883371.29
      1406455.01      6883188.01
#Sta/Elev= 30
  4561.5 2016.48  4581.7 2017.95  4595.6 2017.24  4601.9 2014.02  4632.3 2008.75
  4703.1 2002.71  4784.1 1999.13  4804.3 1996.18  4844.8 1996.15    4865 1993.75
  4985.1 1991.25    5000  1988.4  5005.9 1983.09  5006.4 1982.59  5025.4 1983.09
  5027.6 1990.59  5036.9 1997.78  5051.3 2000.16    5064 1992.43  5073.3    1989
  5079.2 1988.93  5086.9 1992.54  5100.4  1995.5  5109.7 2002.23  5115.6 2004.25
    5158 2014.74  5173.2 2018.27  5188.4 2018.08  5194.4 2020.76  5217.2  2021.4
#Mann= 3 ,-1 , 0
  4561.5     .07       0  5005.9     .07       0  5025.4     .07       0
Bank Sta=5005.9,5025.4
XS Rating Curve= 0 ,0
Exp/Cntr=0.3,0.1

Type RM Length L Ch R = 1 ,12770   ,495,495,495
BEGIN DESCRIPTION:
Bluff Creek 16.0
END DESCRIPTION:
XS GIS Cut Line= 3
      1407155.02      6883288.02      1406985.23      6883158.41
        1406555.        6882938.
#Sta/Elev= 30
  4786.4 2019.93  4789.6 2019.93  4793.7 2017.98    4800 2018.91  4808.2 2018.49
  4822.8 2014.97  4849.9 2012.57  4864.4 2010.53  4872.6 2008.34  4893.5 2005.77
  4964.2 1998.88    4997 1990.13  5002.9 1990.13  5008.9 1988.54  5012.9 1982.68
  5013.4 1982.18  5032.5 1982.68  5036.7 1986.02  5045.2 1990.17  5053.3 1991.15
  5081.1 1992.27  5090.1 1991.47  5186.5 1999.59  5275.3 2003.01  5281.2 2004.45
  5319.7 2005.18  5341.9 2008.17  5348.6 2007.62  5386.3 2009.64  5483.4 2018.99
#Mann= 3 ,-1 , 0
  4786.4     .07       0  5012.9     .07       0  5032.5     .07       0
Bank Sta=5012.9,5032.5
XS Rating Curve= 0 ,0
Exp/Cntr=0.3,0.1

Type RM Length L Ch R = 1 ,12275   ,479,479,479
BEGIN DESCRIPTION:
Bluff Creek 15.0
END DESCRIPTION:
XS GIS Cut Line= 3
      1407354.95        6882788.       1407104.6        6882763.
      1406605.02        6882788.
#Sta/Elev= 30
  4748.4 2020.41  4750.9 2020.41  4758.4 2016.74  4778.5 2011.61  4796.1 2005.93
  4808.7  2003.8  4818.7  2003.2  4828.8 1999.64  4959.4 1988.78  4969.4 1987.53
  4969.7 1983.46  4970.2 1982.96  4989.3 1983.46  4989.5 1984.29  4997.3 1986.92
  5002.3 1986.92  5019.6 1990.69  5039.6 1992.78  5129.8  1994.8  5197.5 1994.37
  5229.9 1996.19  5269.9 1996.92    5310 1999.06    5350 2002.87  5370.1 2003.78
  5390.1 2006.18  5397.6 2008.08  5402.6 2007.46  5440.1  2012.7  5500.2 2016.79
#Mann= 3 ,-1 , 0
  4748.4     .07       0  4969.7     .07       0  4989.3     .07       0
Bank Sta=4969.7,4989.3
XS Rating Curve= 0 ,0
Exp/Cntr=0.3,0.1

Type RM Length L Ch R = 1 ,11796   ,495,495,495
BEGIN DESCRIPTION:
Bluff Creek 14.0
END DESCRIPTION:
XS GIS Cut Line= 3
      1407154.98        6882388.      1406949.79      6882438.43
      1406505.04        6882488.
#Sta/Elev= 30
  4788.7 2008.87    4812 2009.01  4848.4 2003.08  4881.4 2000.48    4890 1996.28
  4895.1 1989.12  4931.5 1987.49  4936.7 1983.87  4943.1 1981.87  4953.9 1981.38
  4954.4 1980.88  4973.5 1981.38  4978.2 1983.99  5024.9 1981.82    5035 1982.45
  5040.6 1985.22  5045.7 1982.32  5085.3  1982.1  5095.4 1984.65  5105.4 1989.75
  5145.7 1989.31  5206.1 1999.35  5226.5 1996.93  5326.8 2008.99  5336.9 2010.97
  5346.9 2015.29    5357 2014.59    5367 2019.06  5402.3  2023.1  5447.5 2025.72
#Mann= 3 ,-1 , 0
  4788.7     .07       0  4953.9     .07       0  4973.5     .07       0
Bank Sta=4953.9,4973.5
XS Rating Curve= 0 ,0
Exp/Cntr=0.3,0.1

Type RM Length L Ch R = 1 ,11301   ,391,391,391
BEGIN DESCRIPTION:
Bluff Creek 13.0
END DESCRIPTION:
XS GIS Cut Line= 3
      1407254.99      6882337.99      1407025.38      6882068.16
      1406805.04        6882038.
#Sta/Elev= 30
  4645.7 2011.29  4652.8 2010.29  4659.4 2010.53  4724.2 2003.41  4816.9 1995.81
  4872.4 1992.38  4886.7  1990.6  4894.4 1991.35  4908.3 1988.95  4921.9 1988.24
  4972.4 1988.76  4982.4 1987.67  4986.7 1987.51  4993.3 1985.69  4996.8 1982.44
  5002.5 1982.44  5010.8 1981.43  5011.3 1980.93  5030.4 1981.43  5036.9 1983.29
  5041.9 1988.01  5060.9 1989.09    5071  1990.8  5075.9 1993.03  5091.2 1998.87
  5101.3 1999.83  5151.8 2008.44  5161.9 2008.92  5181.3 2008.06  5222.4 2010.08
#Mann= 7 ,-1 , 0
  4645.7     .07       0  4816.9     .16       0  4982.4     .07       0
  5002.5     .16       0  5010.8     .07       0  5030.4     .16       0
  5075.9     .07       0
Bank Sta=5010.8,5030.4
XS Rating Curve= 0 ,0
Exp/Cntr=0.3,0.1

Type RM Length L Ch R = 1 ,10910   ,599,599,599
BEGIN DESCRIPTION:
Bluff Creek 12.0
END DESCRIPTION:
XS GIS Cut Line= 3
      1407504.97      6882037.97      1407303.26      6881833.81
      1407055.01        6881738.
#Sta/Elev= 30
    4713 2010.13  4716.5 2010.13    4720 2006.59  4727.1 2004.05  4748.3 2000.62
  4769.5 1999.61  4815.4 1995.63  4889.7 1988.42    4922 1987.14  4946.3 1985.72
  4974.6 1987.75  4981.6 1987.58  4988.7 1985.66    4993 1981.27  4993.5 1980.77
  5012.8 1981.27  5019.6 1984.16  5032.8 1986.74  5051.7 1985.73  5062.8 1989.02
  5094.6 1992.79    5112 1994.08  5117.4 1995.29  5171.9 2000.21  5212.5 2006.54
  5226.5 2009.24    5234 2012.09  5251.1 2012.99  5256.5 2015.14  5266.1 2014.97
#Mann= 5 ,-1 , 0
    4713     .07       0  4815.4     .16       0    4922     .07       0
    4993     .07       0  5012.8     .07       0
Bank Sta=4993,5012.8
XS Rating Curve= 0 ,0
Exp/Cntr=0.3,0.1

Type RM Length L Ch R = 1 ,10311   ,599,599,599
BEGIN DESCRIPTION:
Bluff Creek 11.0
END DESCRIPTION:
XS GIS Cut Line= 3
      1408054.99      6881687.99      1407691.17      6881501.13
      1407504.99      6881137.98
#Sta/Elev= 30
    4591 2010.05  4665.8 2000.76  4754.6 1993.23  4865.5 1990.52  4882.1  1987.1
  4892.9 1986.52  4909.9 1986.78    4917 1988.34  4926.4 1987.05  4932.1 1988.15
  4938.5 1986.42  4970.8 1982.96  4984.5 1983.93    4993 1982.42  4995.3 1980.09
  4995.8 1979.59  5016.4 1980.09  5022.4 1981.47  5028.1 1984.93  5050.2 1982.82
  5066.8 1984.97  5111.2 1985.54  5127.1 1987.07  5149.6 1995.67  5155.6 2000.25
  5161.2 2000.12  5172.1 2004.81  5177.8 2008.73  5250.7 2012.06  5408.1 2012.21
#Mann= 5 ,-1 , 0
    4591     .07       0  4892.9     .16       0  4938.5     .07       0
  4995.3     .07       0  5016.4     .07       0
Bank Sta=4995.3,5016.4
XS Rating Curve= 0 ,0
Exp/Cntr=0.3,0.1

Type RM Length L Ch R = 1 ,9712    ,573,573,573
BEGIN DESCRIPTION:
Bluff Creek 10.0
END DESCRIPTION:
XS GIS Cut Line= 3
      1408304.98      6881437.98      1408048.27      6881094.51
      1407505.01      6880288.02
#Sta/Elev= 30
  4571.2 2011.53  4593.1 2005.34  4607.7 2004.01  4643.1 2004.45  4728.5 1998.61
  4784.8 1991.24  4843.2 1986.21  4978.7 1982.88  4984.9 1982.33    4988  1979.4
  4988.5  1978.9  5009.1  1979.4  5035.3 1984.64  5071.3 1986.36  5086.3    1985
  5092.3 1986.71  5116.3 1984.46  5143.3 1986.21  5188.2 1982.85  5224.2 1986.35
  5230.3  1985.2  5245.2 1987.63  5296.2 1989.69  5446.2 2006.29  5626.1 2016.76
  5791.6 2029.34    5893 2035.18  5928.9 2038.03  5964.9  2042.8  5972.4 2045.19
#Mann= 3 ,-1 , 0
  4571.2     .07       0    4988     .07       0  5009.1     .07       0
#XS Ineff= 2 , 0
                         5067.71         2001.97
Permanent Ineff=
       F       F
Bank Sta=4988,5009.1
XS Rating Curve= 0 ,0
Exp/Cntr=0.3,0.1

Type RM Length L Ch R = 1 ,9139    ,542,542,542
BEGIN DESCRIPTION:
Bluff Creek 9.0
END DESCRIPTION:
XS GIS Cut Line= 6
      1408360.66      6881361.91      1408243.97      6881175.46
      1408378.43      6880999.35      1408414.41      6880902.77
      1408405.37      6880730.18      1408005.01        6880538.
#Sta/Elev= 30
  4219.3 2011.81  4261.7 2005.31  4298.3 2003.95  4319.5  2006.4  4334.8 2004.45
  4350.1 1997.79  4407.9 1989.04  4429.1 1992.42  4594.2 1991.61  4609.4 1989.63
  4630.4 1991.64  4645.6  1989.5  4651.5 1991.61  4667.1 1991.72  4692.1 1989.77
  4747.4 1991.98  4899.2 1991.44  4912.7 1989.76    4980    1991  4995.6 1979.22
  5001.4 1979.79  5006.7 1973.93  5007.2 1973.43  5027.8 1973.93  5034.6 1985.99
  5040.2 1987.17  5144.7 1996.09  5221.8 1999.85  5265.8 2005.28  5386.9 2007.23
#Mann= 3 ,-1 , 0
  4219.3     .07       0  5006.7     .07       0  5027.8     .07       0
Bank Sta=5006.7,5027.8
XS Rating Curve= 0 ,0
Exp/Cntr=0.3,0.1

Type RM Length L Ch R = 1 ,8597    ,573,573,573
BEGIN DESCRIPTION:
Bluff Creek 8.0
END DESCRIPTION:
XS GIS Cut Line= 4
      1409035.13      6880854.06      1408906.35      6880552.43
      1408471.93      6880271.52      1408055.01        6880188.
#Sta/Elev= 30
  4154.7 2004.89  4226.5 2003.41  4267.1 1999.92  4335.3 2000.77    4357 1997.56
  4401.5 1994.58  4501.1 1990.77  4516.3 1992.82  4558.5 1990.85  4609.9 1990.66
  4718.8 1984.81  4805.8 1983.69  4921.3 1979.15  4936.4 1980.15  4984.6 1978.06
  5027.1 1972.34  5027.6 1971.84  5048.3 1972.34  5058.1 1974.69  5078.5 1973.76
  5088.7 1974.84  5099.1 1979.78  5109.1 1987.41  5119.3 1997.92  5129.5 2003.59
    5145 2001.99  5150.1 2004.21  5195.9  2006.2  5241.6 2006.06  5425.2 2015.12
#Mann= 3 ,-1 , 0
  4154.7     .07       0  5027.1     .07       0  5048.3     .07       0
Bank Sta=5027.1,5048.3
XS Rating Curve= 0 ,0
Exp/Cntr=0.3,0.1

Type RM Length L Ch R = 1 ,8024    ,589,589,589
BEGIN DESCRIPTION:
Bluff Creek 7.0
END DESCRIPTION:
XS GIS Cut Line= 3
        1409005.        6880388.      1408860.18      6879988.44
      1408654.99      6879637.99
#Sta/Elev= 30
    4575 1998.72  4590.3 1998.08  4620.9  2001.8  4638.8 1997.64  4682.2 1993.06
  4745.2 1989.47  4763.4 1989.26  4862.2 1982.57  4941.9 1979.24  4967.2 1976.77
  4979.2  1976.6  4986.9  1969.3  4987.4  1968.8  5008.3  1969.3  5012.1 1971.19
  5034.7 1974.56    5105  1976.9  5142.1 1977.17  5163.6 1980.93  5179.3 1987.43
  5185.9 1991.62    5195 1993.28  5200.8 1992.04  5216.5 1997.59  5222.3 1997.53
  5232.2 2001.41  5302.4 2003.59  5333.8 2001.76  5398.2 2000.39  5406.1  1999.4
#Mann= 3 ,-1 , 0
    4575     .07       0  4986.9     .07       0  5008.3     .07       0
Bank Sta=4986.9,5008.3
XS Rating Curve= 0 ,0
Exp/Cntr=0.3,0.1

Type RM Length L Ch R = 1 ,7435    ,595,595,595
BEGIN DESCRIPTION:
Bluff Creek 6.0
END DESCRIPTION:
XS GIS Cut Line= 3
        1409455.      6880037.99      1409261.27      6879686.21
      1408904.99        6879488.
#Sta/Elev= 30
  4598.4  2000.3  4621.2 1994.33  4633.9 1993.68  4666.1 1997.03  4671.8 1993.38
  4678.3 1991.63  4715.3  1989.8  4812.8 1992.53  4818.5 1995.63  4840.3 1998.31
  4878.2 1997.49  4894.2 1994.78  4899.9 1991.44    4916 1990.83  4929.5  1986.4
  4959.6  1982.7  4975.1 1978.35  4987.1 1970.87    5000 1970.13  5007.9 1966.03
  5008.4 1965.53  5029.3 1966.03  5031.5 1971.16  5041.5 1973.17  5110.3 1976.82
  5159.4 1979.22  5188.1    1982    5259 1995.05  5304.7  2001.9  5407.7 1998.74
#Mann= 5 ,-1 , 0
  4598.4     .07       0  5007.9     .07       0  5029.3     .07       0
  5110.3     .16       0  5159.4     .07       0
Bank Sta=5007.9,5029.3
XS Rating Curve= 0 ,0
Exp/Cntr=0.3,0.1

Type RM Length L Ch R = 1 ,6840    ,600,600,600
BEGIN DESCRIPTION:
Bluff Creek 5.0
END DESCRIPTION:
XS GIS Cut Line= 3
      1409854.98      6879787.97      1409410.03      6879143.08
      1408604.96      6878687.98
#Sta/Elev= 30
  4216.5 2005.09    4230 2005.34  4242.2 2001.11  4274.6 1996.28  4374.4 1994.55
  4410.9 1992.01    4424 1988.99  4453.8 1988.15  4525.4 1990.89  4555.2 1996.47
    4591 1998.59  4632.9 1993.68  4647.8 1994.26  4677.6 1988.74  4704.6 1980.81
  4734.4 1977.35  4841.9 1972.28  4939.3 1970.77  4957.6  1967.3  4959.6 1963.68
  4960.1 1963.18    4981 1963.68  5005.8  1979.8  5038.4 1980.65  5074.7 1980.57
  5248.4 1991.52  5540.4 1998.82  5572.8 1999.82    5836 2009.78  5924.8 2015.27
#Mann= 8 ,-1 , 0
  4216.5    .035       0  4242.2     .07       0  4939.3     .16       0
  4959.6     .07       0    4981     .16       0  5038.4     .07       0
  5540.4     .16       0  5572.8     .07       0
Bank Sta=4959.6,4981
XS Rating Curve= 0 ,0
Exp/Cntr=0.3,0.1

Type RM Length L Ch R = 1 ,6240    ,945,945,945
BEGIN DESCRIPTION:
Bluff Creek 4.0
END DESCRIPTION:
XS GIS Cut Line= 3
       1409980.2      6878937.07       1409804.6      6878837.83
        1409455.        6878588.
#Sta/Elev= 30
  4798.3 1994.73  4829.9 1990.26  4845.8 1992.31  4851.6 1990.78  4867.5 1995.49
  4919.1    1985  4923.6 1982.31  4926.7 1980.45  4932.4 1982.15  4942.1 1979.96
  4948.4 1975.17  4954.1 1973.15    4970 1970.42  4976.6 1966.72  4980.9 1961.54
  4981.4 1961.04  5002.4 1961.54  5002.8 1965.13    5007 1968.86  5013.1 1966.65
  5021.7 1969.49  5036.4 1967.26  5042.6 1969.63  5048.8  1968.8  5057.4 1970.89
  5166.4 1971.55  5336.3 1978.45  5365.8 1982.67  5392.8 1990.48  5429.7 1990.86
#Mann= 5 ,-1 , 0
  4798.3     .07       0  4923.6     .16       0  4980.9     .07       0
  5002.4     .16       0  5166.4     .07       0
Bank Sta=4980.9,5002.4
XS Rating Curve= 0 ,0
Exp/Cntr=0.3,0.1

Type RM Length L Ch R = 1 ,5295    ,205,205,205
BEGIN DESCRIPTION:
Bluff Creek 3.0
END DESCRIPTION:
XS GIS Cut Line= 3
      1409976.55      6878726.64      1409944.79       6878137.5
      1409795.97      6877857.83
#Sta/Elev= 30
    4410 1985.93  4448.7 1984.08  4468.7 1984.13  4527.7 1980.98  4568.9 1977.95
    4669 1973.53  4720.8 1972.44  4819.2 1971.83  4903.8 1970.07  4929.4  1968.9
  4939.4 1969.35  4969.5 1967.55  4979.5 1964.95  4986.4 1961.06  4986.9 1960.56
    5008 1961.06  5013.3 1962.35  5029.6 1982.72  5035.3 1984.73  5057.3 1989.31
  5079.2 1988.19  5089.9  1988.7  5139.5 1987.99  5227.4 1989.67  5243.7 1989.23
  5249.3 1989.89  5281.9 1989.89  5287.6 1991.05  5303.9 1990.11  5316.8 1990.85
#Mann= 3 ,-1 , 0
    4410     .07       0  4986.4     .07       0    5008     .07       0
Bank Sta=4986.4,5008
XS Rating Curve= 0 ,0
Exp/Cntr=0.3,0.1

Type RM Length L Ch R = 1 ,5090    ,905,905,905
BEGIN DESCRIPTION:
Bluff Creek 2.0
END DESCRIPTION:
XS GIS Cut Line= 3
      1410160.12      6878663.39      1410150.08      6878138.09
       1410042.1      6877711.96
#Sta/Elev= 30
  4474.6 1988.78    4600 1986.71  4619.7 1987.79    4630 1988.01    4660 1980.19
  4717.8 1976.78    4750 1975.76    4770 1973.73  4800.1 1974.37  4810.1 1972.84
  4830.1 1972.35  4860.1 1972.94  4880.1 1970.77  4940.1 1968.93  4990.1 1964.99
  4997.5 1962.56  5002.8 1962.67  5009.9 1958.81  5010.4 1958.31  5031.5 1958.81
  5038.6 1966.74  5057.2 1968.62  5072.3 1971.26  5084.8 1969.75  5120.6 1973.09
  5144.5 1972.87  5166.7 1975.15  5207.7 1974.36  5379.6 1980.24  5439.6 1980.29
#Mann= 7 ,-1 , 0
  4474.6     .07       0  4619.7    .035       0  4717.8     .07       0
  5009.9     .07       0  5031.5     .07       0  5057.2    .035       0
  5379.6     .07       0
Bank Sta=5009.9,5031.5
XS Rating Curve= 0 ,0
Exp/Cntr=0.3,0.1

Type RM Length L Ch R = 1 ,4185    ,387,387,387
BEGIN DESCRIPTION:
Bluff Creek 1.0
END DESCRIPTION:
XS GIS Cut Line= 3
      1410904.98      6878337.96      1410825.53      6878118.29
      1410055.01      6877338.01
#Sta/Elev= 30
  4766.4 1986.21    4807  1985.8  4893.6 1986.87    4899 1987.89  4936.5 1984.88
  4947.1 1982.46    4955 1972.07  4960.3 1967.15  4968.2 1956.04  4968.7 1955.54
  4989.8 1956.04  4990.9 1959.65  5007.6 1959.59  5021.8 1962.61  5028.8 1966.25
  5035.9 1966.89  5297.5 1969.31  5672.4 1968.73  5728.9 1970.44  5785.5 1975.12
  5820.8 1976.44  5874.4 1980.02  5898.7 1981.85  5926.9 1982.36    5934    1981
  5962.8  1980.8  6011.8 1982.18  6018.8 1984.25  6047.1 1985.55  6096.6 1986.29
#Mann= 5 ,-1 , 0
  4766.4     .07       0  4968.2     .07       0  4989.8     .07       0
  5874.4    .035       0  5962.8     .07       0
Bank Sta=4968.2,4989.8
XS Rating Curve= 0 ,0
Exp/Cntr=0.3,0.1

Type RM Length L Ch R = 1 ,3798    ,715,715,715
BEGIN DESCRIPTION:
Bluff Creek 4278
END DESCRIPTION:
XS GIS Cut Line= 5
      1411076.05       6878181.9      1411072.44      6877755.67
      1410905.21      6877758.05      1410595.01      6877799.07
       1410279.1      6877524.27
#Sta/Elev= 30
  4406.5  1979.5  4480.4 1978.05  4537.3 1975.62  4640.4 1970.55  4680.4 1969.79
  4790.4 1968.88  4820.4 1969.74  4850.2 1968.56  4880.2 1969.44  4940.2 1969.28
  4950.2 1968.41  4960.2 1966.09  4970.2 1961.93  4979.4 1954.69  4979.9 1954.19
  5000.5 1954.19    5001 1954.69  5002.6 1956.44  5010.3 1959.37  5020.4 1961.31
  5041.7 1964.15  5070.8 1965.29  5267.1 1968.48  5455.7 1968.49  5582.9 1966.81
  5611.4 1967.97  5632.3 1967.94    5675 1971.64  5703.5 1975.09  5731.6 1976.33
#Mann= 4 ,-1 , 0
  4406.5    .035       0  4537.3     .07       0  4979.4     .07       0
    5001     .07       0
Bank Sta=4979.4,5001
XS Rating Curve= 0 ,0
Exp/Cntr=0.3,0.1

Type RM Length L Ch R = 1 ,3083    ,382,382,382
BEGIN DESCRIPTION:
Bluff Creek 4277
END DESCRIPTION:
XS GIS Cut Line= 5
      1411115.13      6877736.61      1410815.63      6877421.49
      1410455.99       6877472.6      1410304.21      6877486.57
      1410204.37      6877408.43
#Sta/Elev= 30
    4202  1969.1  4222.4 1967.89  4243.4 1967.76  4300.1 1968.78  4554.8 1968.76
    4697 1968.44  4862.7 1967.33    4900 1966.74  4933.5 1965.24  4950.5 1963.27
  4960.6 1959.79  4969.9 1954.37  4970.4 1953.87  4991.6 1954.37    4998 1960.84
  5005.2 1960.69    5011 1962.63  5021.1 1963.37  5031.1 1962.41  5041.2 1965.64
  5071.3 1959.49  5081.3 1963.65  5101.4 1966.74    5110  1969.1    5115 1969.39
  5121.5 1972.38  5149.5 1978.84  5186.9 1979.23  5256.1  1981.6  5279.2 1982.59
#Mann= 6 ,-1 , 0
    4202     .07       0  4554.8    .035       0    4697     .07       0
  4969.9     .07       0  4991.6     .07       0  5256.1    .035       0
Bank Sta=4969.9,4991.6
XS Rating Curve= 0 ,0
Exp/Cntr=0.3,0.1

Type RM Length L Ch R = 1 ,2701    ,338,338,338
BEGIN DESCRIPTION:
Bluff Creek 4276
END DESCRIPTION:
XS GIS Cut Line= 3
      1410959.59      6877443.16      1410407.33      6877143.96
      1409965.64      6877078.58
#Sta/Elev= 30
  4371.9 1967.89  4416.1 1968.07  4601.6 1966.82  4808.4 1966.18  4961.4 1963.19
  4968.5 1962.05  4977.6 1958.53  4980.4 1952.58  4980.9 1952.08  5002.1 1952.58
  5003.3 1957.14    5007  1959.8  5052.9 1966.22  5071.8 1965.43  5076.5 1962.85
  5083.2 1962.94  5093.3 1960.58  5103.4 1959.98  5113.6 1968.69  5123.7 1974.38
  5133.8 1976.18    5141 1975.73    5146 1973.14    5154 1971.99  5171.5 1972.61
  5184.3 1974.57  5210.5 1975.73  5224.8 1978.49  5265.2 1981.37  5446.5  1988.6
#Mann= 7 ,-1 , 0
  4371.9     .07       0  4416.1    .035       0  4601.6     .07       0
  4980.4     .07       0  5002.1     .07       0  5071.8    .035       0
  5171.5     .07       0
Bank Sta=4980.4,5002.1
XS Rating Curve= 0 ,0
Exp/Cntr=0.3,0.1

Type RM Length L Ch R = 1 ,2363    ,771,771,771
BEGIN DESCRIPTION:
Bluff Creek 4274
END DESCRIPTION:
XS GIS Cut Line= 5
       1411133.2      6877629.77       1411024.7       6877273.9
        1410655.      6876987.98      1410647.09      6876813.83
      1410088.56      6876861.45
#Sta/Elev= 30
  4160.6 1967.38  4486.5 1967.13  4550.8 1964.76  4685.8 1964.19  4714.7 1962.78
  4721.9 1960.78  4729.2 1962.54  4828.8 1961.04  4857.8 1962.37  4913.9 1958.03
  4928.4 1958.34  4936.6 1960.86  4957.4 1959.21  4963.8 1956.55  4967.4 1951.91
  4967.9 1951.41  4989.1 1951.91  4992.7 1956.91  5002.5 1956.44    5010 1960.48
    5060 1967.62  5090.1 1969.13  5278.6 1968.94  5357.1 1968.62  5378.2 1971.61
  5387.2 1972.82  5427.3 1971.96  5467.5 1975.89  5537.7 1979.57  5734.9 1984.85
#Mann= 5 ,-1 , 0
  4160.6     .07       0  4967.4     .07       0  4989.1     .07       0
  5278.6    .035       0  5378.2     .07       0
Bank Sta=4967.4,4989.1
XS Rating Curve= 0 ,0
Exp/Cntr=0.3,0.1

Type RM Length L Ch R = 1 ,1592    ,0,0,0
BEGIN DESCRIPTION:
Bluff Creek 0.1
END DESCRIPTION:
XS GIS Cut Line= 5
        1411205.      6878388.02      1411243.08      6876868.85
      1411155.44      6876832.82      1410894.67      6876743.32
      1410028.24      6876765.09
#Sta/Elev= 30
  3385.6 1982.28  3465.6 1981.63  3835.8 1970.23  3865.8  1971.4  3905.8 1969.73
  4165.9 1966.81  4285.9 1967.07  4315.9 1965.48    4736 1963.62  4905.2 1965.15
  4944.5 1963.21  4967.9 1958.38  4973.3 1959.13  4978.9 1957.42  5002.9 1956.08
  5010.8 1949.86  5011.3 1949.36  5032.5 1949.86  5033.9 1953.37  5059.8 1961.55
  5091.1 1964.46  5193.2 1964.76  5272.9 1966.52  5625.3 1968.62  5675.5 1968.63
  5715.5  1971.5  5755.5 1970.82  5825.5 1976.18  6004.9 1982.28  6142.4  1986.4
#Mann= 7 ,-1 , 0
  3385.6     .07       0  4944.5    .035       0  5010.8    .035       0
  5032.5    .035       0  5193.2     .07       0  5625.3    .035       0
  6004.9     .07       0
Bank Sta=5010.8,5032.5
XS Rating Curve= 0 ,0
Exp/Cntr=0.3,0.1

Chan Stop Cuts=-1
Use User Specified Reach Order=0
Composite Channel Slope=5
