HEC-RAS study Holder Creek.prj: Holder Creek Base Level Engineering

--- Holder Creek.g01 (geometry) --- (continued)

Type RM Length L Ch R = 1 ,37648   ,499,499,499
BEGIN DESCRIPTION:
Holder Creek 60.0
END DESCRIPTION:
XS GIS Cut Line= 3
      1405355.04      6808687.97      1405951.55      6808239.49
      1406104.98      6808088.02
#Sta/Elev= 30
  4253.7 2429.53  4256.8 2429.53  4260.9 2424.37  4310.9 2408.55  4360.9 2403.16
    4690 2402.09  4704.1 2401.71  4731.6 2396.15  4741.1 2396.08  4781.6 2400.57
  4796.2 2400.35  4810.8 2396.33    4917 2399.84  4946.1 2397.62  4960.7 2393.33
    4967 2394.15  4981.5 2392.41  4986.6  2389.2  4987.1  2388.7  5005.7  2389.2
  5010.6 2401.05  5017.7 2414.81  5031.8 2424.62  5038.8 2424.87    5046 2428.35
    5053 2429.57  5060.1 2434.66  5088.4 2441.75  5198.5 2462.57  5215.6 2464.97
#Mann= 5 ,-1 , 0
  4253.7     .07       0  4741.1     .16       0  4986.6     .07       0
  5005.7     .16       0  5198.5     .07       0
Bank Sta=4986.6,5005.7
XS Rating Curve= 0 ,0
Exp/Cntr=0.3,0.1

Type RM Length L Ch R = 1 ,37149   ,497,497,497
BEGIN DESCRIPTION:
Holder Creek 59.0
END DESCRIPTION:
XS GIS Cut Line= 5
      1405305.02      6808787.99      1405610.63      6808634.85
      1405734.69      6808657.87      1405894.48      6808694.75
        1406355.        6808488.
#Sta/Elev= 30
    4532 2463.61  4545.9 2460.42  4568.3 2450.56  4629.7 2417.93  4635.3 2417.08
  4652.1 2409.36  4674.4  2404.2  4719.1 2399.21  4858.8 2400.55  4908.8 2399.08
  4939.3 2394.63  5002.7 2392.14  5021.6  2388.6  5022.1  2388.1  5040.7  2388.6
  5051.6 2391.68  5061.9 2397.55  5067.2 2404.75  5082.4 2411.58  5109.9    2413
  5161.7  2410.6  5201.7 2411.28  5313.7 2414.06  5383.2 2417.72    5435 2422.66
  5481.3 2429.05  5533.1 2443.66  5578.4 2452.22  5608.1 2459.56  5668.8 2467.88
#Mann= 5 ,-1 , 0
    4532     .07       0  5021.6     .07       0  5040.7     .07       0
  5201.7     .16       0  5578.4     .07       0
Bank Sta=5021.6,5040.7
XS Rating Curve= 0 ,0
Exp/Cntr=0.3,0.1

Type RM Length L Ch R = 1 ,36652   ,499,499,499
BEGIN DESCRIPTION:
Holder Creek 58.0
END DESCRIPTION:
XS GIS Cut Line= 3
      1405355.03        6809088.      1405556.65      6809098.68
      1405754.98      6809038.01
#Sta/Elev= 30
  4798.1 2464.84  4818.1 2464.04  4828.1 2462.92  4838.1 2451.03  4848.1 2431.55
  4868.2 2416.99  4878.2 2407.36  4887.9 2401.75  4892.9 2402.35  4898.2 2397.54
  4908.2  2393.4  4918.2  2391.3  4928.2 2390.26  4968.3 2390.82  4978.3 2390.17
  4996.7 2386.91  4999.2 2385.86  4999.7 2385.36  5017.8 2385.36  5018.3 2385.86
  5029.6 2386.96  5049.5 2395.62  5054.7 2393.64    5061 2396.09  5081.9 2398.68
  5092.7 2400.97  5113.3  2402.4  5134.2 2405.07  5158.3 2407.02  5207.4 2408.54
#Mann= 3 ,-1 , 0
  4798.1     .07       0  4999.2     .07       0  5018.3     .07       0
Bank Sta=4999.2,5018.3
XS Rating Curve= 0 ,0
Exp/Cntr=0.3,0.1

Type RM Length L Ch R = 1 ,36153   ,475,475,475
BEGIN DESCRIPTION:
Holder Creek 57.0
END DESCRIPTION:
XS GIS Cut Line= 3
        1405455.        6809488.      1405678.13      6809511.83
        1405805.      6809088.02
#Sta/Elev= 30
  4775.6 2450.22  4786.1 2449.53  4795.7 2448.73  4815.8 2445.54  4826.8 2442.04
  4866.1 2432.35  4906.3 2418.19  4914.1 2414.77  4919.1 2410.22  4926.5 2406.81
  4946.6 2401.17  4966.7 2387.47  4976.7  2386.2  4986.8  2386.1  4995.9 2384.67
  4998.3    2383  4998.8  2382.5  5017.4    2383  5024.9  2384.9  5056.2 2386.04
  5066.6 2388.48  5074.1 2391.19  5107.2 2390.33  5129.3 2391.24  5139.7 2392.86
  5150.7 2395.77  5178.6 2398.34  5321.4 2399.85  5369.3 2402.27  5442.4 2407.43
#Mann= 4 ,-1 , 0
  4775.6     .16       0  4786.1     .07       0  4998.3     .07       0
  5017.4     .07       0
Bank Sta=4998.3,5017.4
XS Rating Curve= 0 ,0
Exp/Cntr=0.3,0.1

Type RM Length L Ch R = 1 ,35678   ,852,852,852
BEGIN DESCRIPTION:
Holder Creek 56.0
END DESCRIPTION:
XS GIS Cut Line= 3
        1406105.      6809737.99      1406145.02      6809538.05
        1406105.      6809238.01
#Sta/Elev= 30
  4796.1 2463.44  4821.6 2461.61  4826.7 2460.13  4845.7 2456.88  4877.7 2449.39
  4887.9 2447.73  4898.1 2446.82  4908.3 2434.54  4918.4 2418.36  4923.5 2418.91
  4928.7  2411.4  4938.9 2404.25  4969.4 2384.25  4974.5 2385.19  4980.2 2379.58
  4980.7 2379.08    4999 2379.08  4999.5 2379.58  5010.1 2381.15  5020.2    2385
  5080.8 2386.28  5109.8 2385.52  5121.1 2384.48  5131.2  2385.3  5151.4 2390.61
  5161.5 2392.58  5171.6 2393.56  5232.1 2394.14  5252.3 2394.86  5302.7 2400.27
#Mann= 4 ,-1 , 0
  4796.1     .16       0  4845.7     .07       0  4980.2     .07       0
  4999.5     .07       0
Bank Sta=4980.2,4999.5
XS Rating Curve= 0 ,0
Exp/Cntr=0.3,0.1

Type RM Length L Ch R = 1 ,34826   ,827,827,827
BEGIN DESCRIPTION:
Holder Creek 54.0
END DESCRIPTION:
XS GIS Cut Line= 3
        1406655.      6809887.99      1406780.01      6809287.97
      1406654.99      6808787.97
#Sta/Elev= 30
  4387.1 2456.38  4438.2  2439.7  4471.8 2424.17  4507.1 2413.96  4540.3  2408.7
  4612.3 2401.59  4657.3 2399.62  4785.4 2382.22  4890.4  2381.3  4952.5 2380.31
  4964.3 2377.49  4979.5 2377.98  4987.8 2372.85  4988.3 2372.35  5007.1 2372.85
  5010.3 2375.99  5020.6 2379.39  5038.7 2382.72  5121.1 2387.29    5250 2388.42
  5298.1 2391.71  5340.1 2395.96  5368.5 2404.74  5373.6 2404.45  5409.7 2420.84
  5414.9 2420.87  5450.9 2436.37  5456.1 2436.12  5476.8 2442.14  5515.4 2447.48
#Mann= 9 ,-1 , 0
  4387.1     .07       0  4471.8     .16       0  4785.4     .07       0
  4890.4     .16       0  4964.3     .07       0  4987.8     .07       0
  5007.1     .07       0  5298.1     .16       0  5476.8     .07       0
Bank Sta=4987.8,5007.1
XS Rating Curve= 0 ,0
Exp/Cntr=0.3,0.1

Type RM Length L Ch R = 1 ,33999   ,496,496,496
BEGIN DESCRIPTION:
Holder Creek 52.0
END DESCRIPTION:
XS GIS Cut Line= 3
        1407855.        6809238.      1407496.82      6809144.04
      1406904.97      6808787.98
#Sta/Elev= 30
  4629.7 2459.96  4632.3 2459.96    4640 2454.21  4647.3 2446.77  4652.5 2445.03
  4681.4 2426.73  4687.7 2420.45  4702.1 2412.24  4722.8 2404.08  4728.1 2398.63
  4741.9 2395.06  4784.8 2385.92    4877 2383.27  4940.7 2378.22  4991.5 2373.81
    5004 2369.57  5004.5 2369.07  5023.6 2369.57  5048.8 2371.19  5063.3 2374.61
  5142.9 2375.08  5195.3 2378.09  5340.6 2379.41  5407.9 2385.62    5444 2390.73
  5523.6 2415.34    5601 2422.94  5655.7 2428.29  5667.4 2431.46  5690.7 2434.17
#Mann= 8 ,-1 , 0
  4629.7     .16       0  4741.9     .07       0    4877     .16       0
  4940.7     .07       0    5004     .07       0  5023.6     .07       0
  5407.9     .16       0    5601     .07       0
Bank Sta=5004,5023.6
XS Rating Curve= 0 ,0
Exp/Cntr=0.3,0.1

Type RM Length L Ch R = 1 ,33503   ,496,496,496
BEGIN DESCRIPTION:
Holder Creek 51.0
END DESCRIPTION:
XS GIS Cut Line= 3
      1407954.99      6809037.98       1407841.8      6808851.66
      1407254.97      6808287.98
#Sta/Elev= 30
    4782 2447.61  4784.9 2447.61  4805.2 2434.42  4832.4 2414.26  4853.7 2394.56
  4875.6 2380.09    4899 2371.89  4948.7 2371.99  4969.8 2366.89  4970.3 2366.39
  4989.4 2366.89  4999.2 2368.89  5042.7 2369.78  5064.1 2372.32  5198.4 2367.74
  5212.5 2370.02  5219.5 2373.18  5281.7 2374.15  5354.1 2376.03  5382.4 2384.45
    5460 2387.73  5580.2 2402.08  5629.8 2410.93  5636.8 2409.75  5640.8 2410.98
  5665.1 2413.34  5707.5 2420.39  5728.9 2428.73    5750 2434.06  5813.7  2441.3
#Mann= 5 ,-1 , 0
    4782     .07       0  4969.8     .07       0  4989.4     .07       0
  5281.7     .16       0  5640.8     .07       0
Bank Sta=4969.8,4989.4
XS Rating Curve= 0 ,0
Exp/Cntr=0.3,0.1

Type RM Length L Ch R = 1 ,33007   ,498,498,498
BEGIN DESCRIPTION:
Holder Creek 50.0
END DESCRIPTION:
XS GIS Cut Line= 3
        1408255.      6808838.05      1408252.95      6808632.16
      1407654.99      6808087.99
#Sta/Elev= 30
  4794.1 2448.55  4818.5 2445.93  4864.2 2441.96  4874.2 2436.51  4904.2  2411.1
  4924.2 2399.48  4974.2 2379.02  4994.2  2374.1  5015.6 2364.66  5019.9 2360.96
  5020.4 2360.46  5039.5 2360.96  5043.9 2365.28  5058.1 2363.39  5086.5 2366.65
  5178.4 2365.34  5232.9 2366.57  5263.5 2366.76  5277.5 2368.45  5291.9  2370.3
  5410.1  2370.9  5536.9 2380.64  5624.4 2383.42    5671 2386.61  5702.1 2389.95
  5737.9 2398.36  5758.8 2406.84  5766.3 2407.19    5773 2410.27  5808.5 2414.97
#Mann= 9 ,-1 , 0
  4794.1     .16       0  4818.5     .07       0  5019.9     .07       0
  5039.5     .07       0  5232.9     .16       0  5277.5     .07       0
  5410.1     .16       0  5536.9     .07       0    5671     .16       0
Bank Sta=5019.9,5039.5
XS Rating Curve= 0 ,0
Exp/Cntr=0.3,0.1

Type RM Length L Ch R = 1 ,32509   ,495,495,495
BEGIN DESCRIPTION:
Holder Creek 49.0
END DESCRIPTION:
XS GIS Cut Line= 3
      1408604.97      6808587.96      1408254.71      6808167.81
        1408155.      6807588.02
#Sta/Elev= 30
    4453 2433.23  4517.4 2417.94  4531.1 2407.12  4552.5 2397.11    4559 2391.13
  4595.5 2377.53  4616.3 2373.06  4765.8  2364.7  4893.6 2365.54  4914.4 2360.42
  4928.7  2361.2  4939.6 2358.15  4940.1 2357.65  4959.5 2358.15  4992.5 2361.85
  5026.5  2359.3  5050.5 2365.57  5070.8 2367.15  5141.3  2367.4  5183.3 2370.97
  5212.9 2374.55  5304.2  2375.9  5365.1 2381.02  5405.7 2391.95    5426 2401.34
    5441 2405.52  5446.3 2410.25  5500.9 2435.74  5507.1 2440.23  5588.3 2465.77
#Mann= 5 ,-1 , 0
    4453     .16       0  4765.8     .07       0  4939.6     .07       0
  4959.5     .07       0  5183.3     .16       0
Bank Sta=4939.6,4959.5
XS Rating Curve= 0 ,0
Exp/Cntr=0.3,0.1

Type RM Length L Ch R = 1 ,32014   ,458,458,458
BEGIN DESCRIPTION:
Holder Creek 48.0
END DESCRIPTION:
XS GIS Cut Line= 3
        1408705.        6808388.      1408578.07      6808211.87
      1408254.98      6807587.96
#Sta/Elev= 30
  4782.9 2420.79  4796.4 2419.82    4805 2414.36  4819.7 2400.42  4840.6 2387.72
  4876.2 2369.13    4897 2361.07  4918.5 2358.36  4947.3 2359.16    4973 2355.28
  4973.5 2354.78  4992.9 2355.28  5013.8  2358.5  5041.5  2355.4  5067.3 2359.03
  5094.4 2364.62  5107.9 2362.77    5162 2365.23  5262.8 2364.65  5364.6 2370.35
  5443.5  2374.4  5506.8 2385.87  5533.6 2396.54  5539.4 2400.69  5561.5 2406.95
  5567.4 2411.99  5600.1 2426.87  5605.8 2427.59  5612.5 2432.17  5702.6  2460.2
#Mann= 7 ,-1 , 0
  4782.9     .16       0    4973     .07       0  4992.9     .16       0
  5067.3     .07       0  5262.8     .16       0  5364.6     .07       0
  5506.8     .16       0
Bank Sta=4973,4992.9
XS Rating Curve= 0 ,0
Exp/Cntr=0.3,0.1

Type RM Length L Ch R = 1 ,31556   ,996,996,996
BEGIN DESCRIPTION:
Holder Creek 47.0
END DESCRIPTION:
XS GIS Cut Line= 3
        1408905.        6808338.      1408985.59      6808108.64
        1408955.        6807488.
#Sta/Elev= 30
  4756.9 2410.26  4767.1 2409.75  4772.4 2406.22  4778.1 2404.64  4841.7 2394.59
    4891 2371.42  4896.3  2372.1  4905.3 2368.83    4922 2365.92  4965.7 2363.84
  4978.7 2361.44    4984 2364.07  4997.7 2356.94  5002.8 2356.94  5010.7 2351.93
  5011.2 2351.43  5030.6 2351.93  5060.7 2354.83  5100.8 2354.54  5114.7  2356.7
  5250.9 2359.92  5395.3 2360.26  5431.2 2360.37  5471.2 2369.91  5501.3 2381.19
  5518.1 2392.12  5523.1 2391.37  5601.4 2444.26  5618.9 2455.12  5621.4 2455.12
#Mann= 5 ,-1 , 0
  4756.9     .16       0  4965.7     .07       0  5010.7     .07       0
  5030.6     .07       0  5395.3     .16       0
Bank Sta=5010.7,5030.6
XS Rating Curve= 0 ,0
Exp/Cntr=0.3,0.1

Type RM Length L Ch R = 1 ,30560   ,491,491,491
BEGIN DESCRIPTION:
Holder Creek 46.0
END DESCRIPTION:
XS GIS Cut Line= 3
      1409105.03      6808337.97      1409682.14      6807713.91
        1409655.      6807488.03
#Sta/Elev= 30
    4150 2394.86  4220.5 2388.94  4259.4 2383.08  4341.2 2377.99  4390.6 2375.77
  4442.1 2370.11    4525 2364.59    4787 2358.17  4843.7  2351.3  4857.9 2353.04
  4899.8 2351.64  4921.4 2352.85    4967 2352.04  4984.9 2351.81  4988.5 2348.41
    4989 2347.91  5008.4 2348.41  5014.5 2352.73  5019.5 2350.46  5026.1 2354.45
  5106.7 2356.79  5126.8 2362.85    5157 2381.68  5167.1 2391.54  5177.2 2398.64
  5183.9 2405.37  5188.9 2402.82  5207.4 2425.37  5217.5 2439.25  5227.5 2441.91
#Mann= 7 ,-1 , 0
    4150     .16       0  4259.4     .07       0  4341.2     .16       0
  4442.1     .07       0    4967     .16       0  4988.5     .07       0
  5008.4     .16       0
Bank Sta=4988.5,5008.4
XS Rating Curve= 0 ,0
Exp/Cntr=0.3,0.1

Type RM Length L Ch R = 1 ,30069   ,498,498,498
BEGIN DESCRIPTION:
Holder Creek 45.0
END DESCRIPTION:
XS GIS Cut Line= 3
      1410205.01      6808538.02      1410061.21       6807930.2
      1410004.99      6807637.96
#Sta/Elev= 30
  4375.4 2418.91  4416.5  2407.8  4436.3 2400.54  4478.2 2383.37  4483.7 2378.74
  4488.8 2378.82  4539.8 2366.33  4568.2 2362.43  4573.3 2363.42    4588 2361.69
  4700.2  2355.9  4724.8 2356.45    4827  2352.9  4958.9 2353.28  4971.4 2352.69
  4996.9 2345.07  4997.4 2344.57  5016.9 2345.07  5032.8 2348.73  5066.2 2349.38
  5167.7 2347.98  5195.7 2353.02  5214.6  2362.2  5219.7  2362.3  5226.3 2369.16
  5266.5 2399.76  5271.6 2398.04  5277.2 2405.69  5287.4 2413.27  5297.6 2414.43
#Mann= 5 ,-1 , 0
  4375.4     .16       0    4588     .07       0  4996.9     .07       0
  5016.9     .07       0  5066.2     .16       0
Bank Sta=4996.9,5016.9
XS Rating Curve= 0 ,0
Exp/Cntr=0.3,0.1

Type RM Length L Ch R = 1 ,29571   ,598,598,598
BEGIN DESCRIPTION:
Holder Creek 44.0
END DESCRIPTION:
XS GIS Cut Line= 3
      1410254.99      6808438.04      1410420.43       6807837.1
        1410155.        6807438.
#Sta/Elev= 30
  4376.7 2391.01  4387.1 2384.93  4393.9 2377.26  4407.9 2369.61    4439  2359.1
  4459.7 2354.98  4500.5 2351.82    4812 2350.56  4886.7  2349.4  4988.7 2345.87
  4999.2  2342.2  5017.9 2340.85  5023.9 2343.04    5037 2340.45  5037.5 2339.95
    5057 2340.45    5075 2341.26    5083 2343.68    5090 2348.98    5096 2346.35
  5105.1 2351.42  5111.1 2349.22    5119 2351.24  5147.1 2347.86  5240.3 2361.82
  5335.2 2371.85  5357.6 2377.66  5420.7  2401.8  5450.7 2408.21  5479.3 2410.64
#Mann= 6 ,-1 , 0
  4376.7     .16       0  4500.5     .07       0    4812     .16       0
  4886.7     .07       0    5037     .07       0    5057     .07       0
Bank Sta=5037,5057
XS Rating Curve= 0 ,0
Exp/Cntr=0.3,0.1

Type RM Length L Ch R = 1 ,28973   ,598,598,598
BEGIN DESCRIPTION:
Holder Creek 43.0
END DESCRIPTION:
XS GIS Cut Line= 3
      1410554.99      6808538.02      1410705.81      6808126.06
      1411104.99      6807638.01
#Sta/Elev= 30
  4561.3 2436.87    4564 2436.87  4571.3 2429.81  4576.6 2421.72  4582.6    2407
  4601.8 2391.27  4607.1 2390.07  4614.6 2382.54  4632.3 2369.32  4637.6  2367.6
  4657.2 2356.19  4662.8 2351.43  4699.8 2346.99  4865.8 2347.39  4944.7  2340.2
  4976.6 2341.02  4987.8 2338.87  5011.7 2339.81  5014.8 2338.34  5015.3 2337.84
  5037.5 2338.34  5040.5 2342.92  5069.2  2348.3  5119.7 2348.81  5161.8    2348
  5196.9 2351.35    5290 2353.07  5481.2 2358.25  5509.9 2360.95  5630.5 2365.18
#Mann= 5 ,-1 , 0
  4561.3     .07       0  5014.8     .07       0  5037.5     .07       0
  5119.7     .16       0    5290     .07       0
Bank Sta=5014.8,5037.5
XS Rating Curve= 0 ,0
Exp/Cntr=0.3,0.1

Type RM Length L Ch R = 1 ,28375   ,558,558,558
BEGIN DESCRIPTION:
Holder Creek 42.0
END DESCRIPTION:
XS GIS Cut Line= 3
      1410654.96      6808638.01      1411074.87      6808558.31
      1411492.48      6807007.56
#Sta/Elev= 30
  4572.6 2414.06  4603.9 2409.97    4651 2393.89  4656.1 2397.39  4703.3  2404.7
  4708.4 2407.96  4728.6 2408.52  4755.6 2406.31  4760.6 2408.61  4806.7 2400.51
    4818 2395.69  4865.2 2359.02    4878 2353.04  4963.4 2335.39  4963.9 2334.89
  4986.1 2335.39    4990 2338.28    5023 2337.89  5041.8 2341.36  5132.4 2343.69
  5594.1 2350.28  5606.8 2350.79  5825.5 2361.99  6059.9 2366.89  6210.9 2373.83
    6357 2393.34  6460.6  2417.3  6478.6 2424.13  6518.5 2430.85    6606 2434.68
#Mann= 7 ,-1 , 0
  4572.6     .16       0  4728.6     .07       0  4963.4     .07       0
  4986.1     .07       0  5594.1     .16       0  5606.8     .07       0
  6210.9     .16       0
Bank Sta=4963.4,4986.1
XS Rating Curve= 0 ,0
Exp/Cntr=0.3,0.1

Type RM Length L Ch R = 1 ,27817   ,599,599,599
BEGIN DESCRIPTION:
Holder Creek 41.0
END DESCRIPTION:
XS GIS Cut Line= 3
      1411004.99      6809438.01      1411553.52      6808684.39
      1411812.64      6807244.52
#Sta/Elev= 30
  4067.9  2436.7  4140.2 2425.95  4166.5 2418.96  4225.9 2408.85  4282.3 2389.59
  4332.6 2379.12  4389.5 2369.83  4460.6 2363.45  4550.3    2359    4659 2354.04
  4808.9    2345  4871.1 2343.62  4947.6 2341.44  4956.1 2336.71    4980 2332.04
  4980.5 2331.54  5003.3 2332.04  5020.2 2335.33  5240.2 2336.46  5270.7 2341.24
  5636.5 2340.27  5666.9 2344.59  5687.3 2342.91  5772.1 2348.66  5819.3 2354.81
  6007.9 2364.33  6317.2 2386.08  6357.9 2394.58  6408.7 2410.48    6463 2420.32
#Mann= 11 ,-1 , 0
  4067.9     .16       0  4166.5     .07       0  4460.6     .16       0
  4550.3     .07       0    4659     .16       0  4808.9     .07       0
  4871.1     .16       0    4980     .07       0  5003.3     .16       0
  5020.2     .07       0  6007.9     .16       0
Bank Sta=4980,5003.3
XS Rating Curve= 0 ,0
Exp/Cntr=0.3,0.1

Type RM Length L Ch R = 1 ,27218   ,585,585,585
BEGIN DESCRIPTION:
Holder Creek 40.0
END DESCRIPTION:
XS GIS Cut Line= 3
        1411505.        6809138.      1411925.06       6808387.8
      1412354.96      6808088.03
#Sta/Elev= 30
  4140.2 2350.53  4199.2  2348.1  4337.7 2342.39    4593 2341.34  4712.7 2341.76
  4780.6  2340.3  4845.7 2336.07  4899.1 2335.44  4942.5  2333.3  4985.3 2324.01
  4985.8 2323.51  5008.7 2324.01  5063.9 2331.05  5093.6 2340.12  5144.2 2340.74
  5236.7 2349.66  5293.4 2358.55  5329.1 2366.09  5352.7 2375.26  5358.8 2376.12
  5388.5 2392.92  5394.6 2394.81  5409.4 2404.39  5415.5 2405.96  5424.3 2412.18
  5430.4 2413.02  5438.8 2417.16  5445.2 2422.12  5501.7 2443.41  5524.1 2446.99
#Mann= 8 ,-1 , 0
  4140.2     .16       0  4199.2     .07       0    4593     .16       0
  4712.7     .07       0  4899.1     .16       0  4985.3     .07       0
  5008.7     .16       0  5501.7     .07       0
Bank Sta=4985.3,5008.7
XS Rating Curve= 0 ,0
Exp/Cntr=0.3,0.1

Type RM Length L Ch R = 1 ,26633   ,596,596,596
BEGIN DESCRIPTION:
Holder Creek 39.0
END DESCRIPTION:
XS GIS Cut Line= 3
      1411355.02      6809537.98      1412140.52       6808724.8
      1412505.03      6808537.98
#Sta/Elev= 30
  3869.4 2376.98  4067.3 2360.46  4378.5 2343.01  4607.2 2339.18  4845.2 2339.28
  4934.4 2337.44  4951.5 2330.69  4958.4 2326.49  4960.9 2322.58  4961.4 2322.08
  4984.3 2322.58  4999.6 2327.62  5016.3 2328.98  5090.5 2330.11  5162.7 2334.26
  5201.5 2346.69  5218.1 2361.01  5223.7 2361.97  5229.8 2370.03  5240.3 2378.98
  5245.9 2378.57  5252.2 2388.16  5262.5 2396.01  5268.1 2398.12  5284.7 2429.76
  5290.3 2426.56  5297.2 2440.99  5306.9  2446.7  5322.3 2449.23  5409.6 2447.51
#Mann= 7 ,-1 , 0
  3869.4     .07       0  4378.5     .16       0  4607.2     .07       0
  4934.4     .16       0  4960.9     .07       0  4984.3     .16       0
  5322.3     .07       0
Bank Sta=4960.9,4984.3
XS Rating Curve= 0 ,0
Exp/Cntr=0.3,0.1

Type RM Length L Ch R = 1 ,26037   ,598,598,598
BEGIN DESCRIPTION:
Holder Creek 38.0
END DESCRIPTION:
XS GIS Cut Line= 3
        1411655.        6809988.      1412456.33      6809177.45
      1412605.01      6808787.96
#Sta/Elev= 30
  3860.2  2416.6    3945 2405.23  4008.7 2385.81  4051.1 2369.72  4157.2 2355.25
  4270.3  2347.8  4701.7 2337.54  4758.3  2333.5  4779.4 2328.82  4863.8 2327.11
  4896.6 2326.35  4970.4 2325.85  5001.1  2320.5  5001.6    2320  5024.6  2320.5
  5037.6 2325.41  5042.9 2330.86  5052.9  2332.4  5152.5  2335.6  5170.7 2338.24
  5207.3 2354.94  5214.3 2361.33  5270.8 2401.52  5277.7 2406.55  5299.1 2433.51
  5341.7 2428.99  5384.7 2415.58  5401.8 2420.18  5407.2 2417.09  5416.9 2418.48
#Mann= 7 ,-1 , 0
  3860.2     .07       0  4863.8     .16       0  4896.6     .07       0
  5001.1     .07       0  5024.6     .07       0  5214.3     .16       0
  5270.8     .07       0
Bank Sta=5001.1,5024.6
XS Rating Curve= 0 ,0
Exp/Cntr=0.3,0.1

Type RM Length L Ch R = 1 ,25439   ,486,486,486
BEGIN DESCRIPTION:
Holder Creek 37.0
END DESCRIPTION:
XS GIS Cut Line= 3
        1412505.      6810488.05      1412506.43      6809727.55
      1413155.01      6808937.98
#Sta/Elev= 30
  4239.5 2430.48  4319.5 2414.57  4409.5 2402.22  4439.5 2392.96  4499.5 2380.65
  4837.3 2339.62  4869.5 2336.89  4889.5 2331.77  4919.5 2332.16  4947.5 2326.84
  4979.5 2323.37  4993.9 2318.12  4994.4 2317.62  5017.7 2318.12  5020.1 2321.22
  5034.2 2319.44  5077.1 2324.81  5133.5 2323.21    5183 2329.36  5253.2 2327.69
  5283.4 2325.94  5317.4  2328.7  5510.1 2329.43  5744.8 2342.04  5808.7 2342.55
  5872.5 2346.38  5896.7 2351.33  5929.9 2361.83  6000.3 2400.79  6021.8  2405.9
#Mann= 10 ,-1 , 0
  4239.5     .07       0  4837.3     .16       0  4947.5     .07       0
  4993.9     .07       0  5017.7     .07       0  5034.2     .16       0
  5253.2     .07       0  5317.4     .16       0  5510.1     .07       0
  5896.7     .16       0
Bank Sta=4993.9,5017.7
XS Rating Curve= 0 ,0
Exp/Cntr=0.3,0.1

Type RM Length L Ch R = 1 ,24953   ,710,710,710
BEGIN DESCRIPTION:
Holder Creek 36.0
END DESCRIPTION:
XS GIS Cut Line= 3
      1412704.99      6810538.03      1412865.44        6809989.
        1413255.        6808788.
#Sta/Elev= 30
    4428 2429.06  4555.5 2403.24  4667.7 2374.53  4733.2  2365.6  4928.1 2352.93
  4944.3 2341.31  4949.5 2349.09  4977.8 2326.99    4983 2330.49  4998.6 2314.38
  4999.1 2313.88  5022.4 2314.38  5042.5  2319.2    5117 2317.23  5143.7 2321.11
  5221.8 2319.08  5262.3 2322.06  5326.9 2319.64  5358.5 2323.52  5523.5 2325.63
  5638.1 2325.97  5738.6 2329.75  5926.9 2338.78  5947.2 2342.31  5984.5 2358.78
  6031.3 2383.32  6049.5 2396.91  6094.4 2414.24  6157.5 2425.64  6262.6 2433.61
#Mann= 8 ,-1 , 0
    4428     .07       0  4998.6     .07       0  5022.4     .07       0
  5262.3     .16       0  5523.5     .07       0  5638.1     .16       0
  5738.6     .07       0  5984.5     .16       0
Bank Sta=4998.6,5022.4
XS Rating Curve= 0 ,0
Exp/Cntr=0.3,0.1

Type RM Length L Ch R = 1 ,24243   ,589,589,589
BEGIN DESCRIPTION:
Holder Creek 35.0
END DESCRIPTION:
XS GIS Cut Line= 3
      1413605.01      6810288.02      1413440.02      6809738.04
      1413254.99      6808937.96
#Sta/Elev= 30
  4425.8 2422.43  4457.1 2415.38  4508.5  2394.9  4530.2 2372.71  4546.8 2360.47
  4603.3 2340.74  4651.2 2332.67  4697.3 2329.12  4835.3 2324.95    4836 2324.92
  4937.4 2324.14  4964.4 2316.48  4979.2 2315.87  4985.4 2312.08  4985.9 2311.58
  5009.4 2312.08  5010.3 2314.48  5045.3 2318.58  5076.6 2318.88    5115 2318.56
  5318.2 2321.54  5605.6 2330.57  5626.4 2334.79  5656.9 2345.72  5699.7 2369.15
  5706.7 2373.82  5711.8 2373.58  5754.5 2399.92  5759.6  2398.6  5821.2 2417.19
#Mann= 8 ,-1 , 0
  4425.8     .07       0  4835.3     .16       0    4836     .07       0
  4985.4     .07       0  5009.4     .07       0  5076.6     .16       0
    5115     .07       0  5699.7     .16       0
Bank Sta=4985.4,5009.4
XS Rating Curve= 0 ,0
Exp/Cntr=0.3,0.1

Type RM Length L Ch R = 1 ,23654   ,600,600,600
BEGIN DESCRIPTION:
Holder Creek 34.0
END DESCRIPTION:
XS GIS Cut Line= 3
      1414105.01      6810088.03      1413971.48      6809570.89
        1413505.        6808888.
#Sta/Elev= 30
  4465.9 2417.31  4468.5 2417.31  4476.3 2400.84  4483.7 2381.29  4488.8 2382.11
  4524.3 2351.68  4529.5 2351.62    4565 2332.69  4589.9  2326.4  4610.8 2322.86
  4662.2 2320.16  4920.4 2318.01    4941 2315.84    4960  2310.5  4960.5    2310
    4984  2310.5  5077.9  2316.2  5230.3 2317.03    5317 2321.51  5517.5 2326.11
  5553.4 2330.28  5602.7  2341.4  5625.2 2344.69  5646.1 2351.37    5676 2367.18
    5682 2368.49  5690.9 2375.27  5711.9 2382.97  5726.8 2393.47    5827 2420.06
#Mann= 4 ,-1 , 0
  4465.9     .07       0    4960     .07       0    4984     .07       0
  5602.7     .16       0
Bank Sta=4960,4984
XS Rating Curve= 0 ,0
Exp/Cntr=0.3,0.1

Type RM Length L Ch R = 1 ,23054   ,774,774,774
BEGIN DESCRIPTION:
Holder Creek 33.0
END DESCRIPTION:
XS GIS Cut Line= 3
      1414404.99      6810088.03      1414544.32      6809486.35
      1413754.97      6808837.97
#Sta/Elev= 30
  4382.4 2411.85  4392.7 2410.44  4401.2 2404.02  4406.3 2408.57  4413.2 2401.04
  4423.5 2396.33  4443.9 2379.06    4449 2379.67  4454.3 2373.27  4491.7 2348.19
  4556.9 2320.73  4587.7 2314.59  4618.5 2311.78  4667.6 2310.96  4885.4 2313.71
  4916.2 2311.52  4967.5 2312.22  4981.9 2311.33  4993.4 2305.75  4993.9 2305.25
  5017.4 2305.75  5026.3 2309.19  5062.8 2308.24    5114 2312.12  5240.1 2309.84
  5295.2 2313.53  5651.9 2329.37  5879.1 2345.77  5971.2 2355.88  6021.5 2372.96
#Mann= 5 ,-1 , 0
  4382.4     .07       0  4993.4     .07       0  5017.4     .07       0
    5114     .16       0  5295.2     .07       0
Bank Sta=4993.4,5017.4
XS Rating Curve= 0 ,0
Exp/Cntr=0.3,0.1

Type RM Length L Ch R = 1 ,22280   ,421,421,421
BEGIN DESCRIPTION:
Holder Creek 32.0
END DESCRIPTION:
XS GIS Cut Line= 3
      1414805.02      6810087.96      1415096.85      6809431.95
      1415355.01      6808787.96
#Sta/Elev= 30
    4282 2410.42  4348.3 2396.06  4366.1  2379.8  4371.5 2378.58  4389.3 2357.93
  4394.8 2357.06  4424.2 2337.28  4464.5 2318.32  4487.8 2311.02  4522.7 2307.13
  4603.5 2306.72  4636.3 2306.06  4904.8 2307.16  4927.7 2304.23    4980 2305.62
  4995.9 2301.76  4996.4 2301.26  5022.2 2301.76  5025.8 2304.68  5079.7 2307.62
  5087.1 2312.58  5101.2 2314.49  5278.1 2314.41  5325.5 2317.85  5434.1 2334.27
  5487.9 2348.92  5600.9 2400.15  5661.6 2430.77    5679 2441.58  5693.8 2446.64
#Mann= 7 ,-1 , 0
    4282     .07       0  4603.5     .12       0  4636.3     .07       0
  4995.9     .07       0  5022.2     .07       0  5325.5     .16       0
  5661.6     .07       0
Bank Sta=4995.9,5022.2
XS Rating Curve= 0 ,0
Exp/Cntr=0.3,0.1

Type RM Length L Ch R = 1 ,21859   ,578,578,578
BEGIN DESCRIPTION:
Holder Creek 31.0
END DESCRIPTION:
XS GIS Cut Line= 3
      1415005.01      6810137.99      1415255.06      6809792.97
      1415604.98      6808988.04
#Sta/Elev= 30
  4573.9 2402.09  4623.3 2394.37  4639.3 2379.75  4667.1 2353.68  4673.2 2351.65
  4709.7 2325.62  4746.7 2311.99    4824 2300.97  4928.6 2303.38  4986.8 2298.64
  4987.3 2298.14  5013.1 2298.64  5017.1 2301.77  5035.1 2302.69  5040.5  2305.6
  5087.4 2305.03  5139.8 2309.87  5430.7 2311.11  5489.8 2313.75    5507 2308.63
  5536.7 2307.38  5572.4 2313.91  5641.4 2315.12    5683 2321.27  5717.2 2329.65
  5740.6 2338.67  5764.1 2352.73    5793  2363.9  5839.9 2389.73  5877.7 2404.71
#Mann= 6 ,-1 , 0
  4573.9     .07       0  4639.3     .12       0  4928.6     .07       0
  4986.8     .07       0  5013.1     .07       0    5683     .16       0
Bank Sta=4986.8,5013.1
XS Rating Curve= 0 ,0
Exp/Cntr=0.3,0.1

Type RM Length L Ch R = 1 ,21281   ,568,568,568
BEGIN DESCRIPTION:
Holder Creek 30.0
END DESCRIPTION:
XS GIS Cut Line= 3
      1415004.99        6810238.      1415428.12      6810311.73
      1416205.01      6809487.99
#Sta/Elev= 30
  4570.5 2407.64  4631.4 2405.83  4657.3 2399.53  4716.9 2398.45  4793.8 2391.56
    4804    2389    4831  2369.2  4836.1 2371.33  4854.7 2361.86  4890.6 2339.13
  4895.7 2341.06  4915.9 2331.66  4945.1 2316.69  4950.2 2320.98  4960.9 2309.02
  4982.7 2295.81  4983.2 2295.31  5009.1 2295.81  5014.7 2297.99    5043 2296.22
  5071.3 2300.95  5240.8  2300.2  5644.2 2306.11  5806.8 2311.33  5849.3 2318.49
  5920.1 2316.69  5941.1 2312.66  5969.4 2317.46  6080.4 2320.05  6132.3 2324.64
#Mann= 6 ,-1 , 0
  4570.5     .07       0  4915.9     .12       0  4960.9     .07       0
  4982.7     .07       0  5009.1     .07       0  6080.4     .16       0
Bank Sta=4982.7,5009.1
XS Rating Curve= 0 ,0
Exp/Cntr=0.3,0.1

Type RM Length L Ch R = 1 ,20713   ,565,565,565
BEGIN DESCRIPTION:
Holder Creek 29.0
END DESCRIPTION:
XS GIS Cut Line= 3
      1415555.02      6810737.99      1415915.05      6810537.89
      1416654.98      6809888.02
#Sta/Elev= 30
  4588.1 2327.34  4883.2 2306.97  4910.6 2300.35  4926.7 2299.29  4932.4 2296.47
  4978.4 2292.45  4978.9 2291.95  5005.3 2292.45  5056.4 2296.76  5063.9  2295.7
  5092.4 2297.18  5127.5 2295.93  5340.1 2296.11  5495.7 2299.25  5605.3 2298.62
  5658.9 2302.97  5701.6 2311.03  5744.3 2322.56  5750.9 2327.45  5779.4 2338.04
    5786 2343.55  5807.9 2354.07  5814.5    2360  5822.1 2363.65  5864.8 2393.15
  5899.9  2419.5  5920.8 2432.86  5931.9 2438.08  5956.8 2448.33  5984.8 2450.63
#Mann= 5 ,-1 , 0
  4588.1     .07       0  4978.4     .07       0  5005.3     .07       0
  5605.3     .16       0  5931.9     .07       0
Bank Sta=4978.4,5005.3
XS Rating Curve= 0 ,0
Exp/Cntr=0.3,0.1

Type RM Length L Ch R = 1 ,20148   ,1183,1183,1183
BEGIN DESCRIPTION:
Holder Creek 28.0
END DESCRIPTION:
XS GIS Cut Line= 3
      1415705.01      6811087.99      1416420.37      6810537.76
      1416654.99      6809938.02
#Sta/Elev= 30
  4097.5 2325.01  4247.9    2319  4297.8 2313.26  4432.8 2305.49  4617.6 2298.13
  4781.6 2295.74  4816.9 2292.65  4917.5 2292.96  4975.7 2287.47  4976.2 2286.97
  5002.7 2287.47  5010.5 2293.24  5231.9 2295.01  5311.1 2295.22  5343.4 2297.72
  5387.5 2312.76  5406.6 2315.76  5411.9 2318.87  5460.9 2333.17  5472.2 2340.98
  5515.1 2363.28  5525.9  2373.8    5545 2385.64  5550.3 2391.66  5568.9 2402.56
  5580.2 2415.87  5596.1 2423.42  5611.8 2435.12  5629.1 2444.15    5644 2448.31
#Mann= 5 ,-1 , 0
  4097.5     .07       0  4975.7     .07       0  5002.7     .07       0
  5231.9     .16       0  5596.1     .07       0
Bank Sta=4975.7,5002.7
XS Rating Curve= 0 ,0
Exp/Cntr=0.3,0.1

Type RM Length L Ch R = 1 ,18965   ,593,593,593
BEGIN DESCRIPTION:
Holder Creek 27.0
END DESCRIPTION:
XS GIS Cut Line= 3
      1416204.99        6811288.      1417021.88      6811121.42
      1417354.99      6810788.01
#Sta/Elev= 30
  4166.3 2308.35  4503.1  2298.3  4564.3 2293.82  4590.8 2289.18    4867 2288.81
  4911.3 2289.12  4939.5 2284.29  4953.8 2284.84  4972.6 2285.13  4976.4  2281.5
  4976.9    2281  5003.5  2281.5    5070 2288.91  5195.5  2288.3  5223.8 2290.46
  5259.2 2302.04  5266.3 2308.39  5273.3 2310.05  5280.4  2317.1  5301.6 2327.87
  5308.7 2333.86  5315.8 2333.31  5322.8  2341.1  5329.9 2338.41    5337 2343.59
    5344  2343.8  5365.3 2352.75  5386.5 2356.58  5414.8 2367.97  5471.3 2381.55
#Mann= 6 ,-1 , 0
  4166.3     .07       0    4867     .16       0  4953.8     .12       0
  4976.4     .07       0  5003.5     .12       0    5070     .16       0
Bank Sta=4976.4,5003.5
XS Rating Curve= 0 ,0
Exp/Cntr=0.3,0.1

Type RM Length L Ch R = 1 ,18372   ,597,597,597
BEGIN DESCRIPTION:
Holder Creek 26.0
END DESCRIPTION:
XS GIS Cut Line= 3
      1416355.04      6812437.97      1417134.82      6811668.08
      1417904.97      6811238.01
#Sta/Elev= 30
  3904.2 2346.46  3917.3 2344.69  4066.8 2334.75  4109.2 2328.04  4165.8 2309.47
  4321.4 2298.08  4646.7 2289.74    4781 2281.45  4938.4  2284.8    4979 2283.45
  4983.1 2277.73  4983.6 2277.23  5010.2 2277.73  5013.2    2281  5028.4 2282.36
  5332.4 2281.14    5376 2283.33  5419.5 2295.02  5441.2 2293.55    5490 2300.83
  5595.8 2312.63  5625.1 2311.42  5662.8 2320.57  5698.9 2320.21  5737.5  2335.5
  5765.6 2350.18    5793 2373.13    5809 2381.02  5872.1 2395.86  5882.1 2396.27
#Mann= 10 ,-1 , 0
  3904.2    .035       0  3917.3     .07       0  4938.4     .16       0
  4983.1     .07       0  5010.2     .16       0  5013.2     .07       0
  5028.4     .16       0    5490     .07       0  5737.5     .16       0
  5872.1     .07       0
Bank Sta=4983.1,5010.2
XS Rating Curve= 0 ,0
Exp/Cntr=0.3,0.1

Type RM Length L Ch R = 1 ,17775   ,1195,1195,1195
BEGIN DESCRIPTION:
Holder Creek 25.0
END DESCRIPTION:
XS GIS Cut Line= 3
      1416804.96      6812538.03      1417610.94      6811946.42
      1418205.03        6811838.
#Sta/Elev= 30
  4000.2    2308    4344 2288.92  4526.8  2284.3  4580.2 2282.86  4630.3 2274.21
  4652.1    2273  4652.6  2272.5  4679.5    2273  4680.5 2275.33  4686.7  2276.5
  4707.6 2277.65  4880.2 2280.51  4952.2 2280.01  4987.7 2273.86  5019.2  2279.1
  5168.1 2278.37  5209.3 2280.41  5227.8 2287.35  5288.8 2297.35  5412.4 2310.53
  5440.6 2320.09  5460.6  2327.4  5481.9 2329.34  5502.2 2336.93  5542.9 2356.75
  5569.9  2376.8  5572.2 2378.65  5577.2 2377.18  5583.5 2387.75  5603.9 2394.54
#Mann= 9 ,-1 , 0
  4000.2     .07       0  4526.8     .16       0  4652.1     .07       0
  4679.5     .16       0  4880.2     .07       0  5168.1     .16       0
  5209.3     .07       0  5440.6     .16       0  5569.9     .07       0
Bank Sta=4652.1,4679.5
XS Rating Curve= 0 ,0
Exp/Cntr=0.3,0.1

Type RM Length L Ch R = 1 ,16580   ,598,598,598
BEGIN DESCRIPTION:
Holder Creek 24.0
END DESCRIPTION:
XS GIS Cut Line= 3
      1416555.01      6813087.99      1417360.46      6812690.48
      1418154.96      6812138.03
#Sta/Elev= 30
  4101.8 2389.81  4132.7 2387.05  4146.4 2382.92  4183.1 2365.33    4191 2357.96
    4200 2353.58  4222.5 2347.03  4250.5 2344.87  4312.3  2333.7  4357.2 2331.16
  4385.2 2335.68    4447 2335.55  4469.4 2331.77  4525.5 2311.26  4570.4 2303.23
  4920.4 2287.33    4952 2285.04  4982.8 2271.55  4985.8  2265.4  4986.3  2264.9
  5013.6  2265.4  5027.2 2269.64    5063 2273.45  5274.9 2273.54  5529.3 2276.03
  5572.8 2281.17  5763.4  2285.1  5820.7 2288.06  5898.4 2295.17  5967.7 2308.19
#Mann= 8 ,-1 , 0
  4101.8     .07       0  4920.4     .16       0  4985.8     .07       0
  5013.6     .16       0  5274.9     .07       0  5763.4     .16       0
  5820.7     .07       0  5898.4     .16       0
Bank Sta=4985.8,5013.6
XS Rating Curve= 0 ,0
Exp/Cntr=0.3,0.1

Type RM Length L Ch R = 1 ,15982   ,599,599,599
BEGIN DESCRIPTION:
Holder Creek 23.0
END DESCRIPTION:
XS GIS Cut Line= 3
      1417204.97      6813138.02      1417844.22      6812728.28
      1418304.98      6812038.03
#Sta/Elev= 30
  4240.7 2325.98  4290.6 2305.24  4342.2 2299.54  4560.3 2288.53  4763.2 2270.59
  4841.8  2271.5    4972 2267.34  4993.1 2263.86  4994.4 2261.17  4994.9 2260.67
  5022.3 2261.17  5023.4  2265.4  5036.4 2272.33  5122.5    2273  5377.3 2285.36
  5498.2 2291.78  5621.2 2300.91  5658.4 2309.08  5678.2 2314.06  5693.3 2322.54
  5714.3 2328.34  5729.3 2339.11  5735.3 2339.88  5744.3    2348  5750.3 2349.47
  5771.4 2361.97  5780.4  2370.7  5801.5  2381.8  5816.4 2391.83  5829.9 2395.06
#Mann= 7 ,-1 , 0
  4240.7     .07       0  4994.4     .07       0  5022.3     .16       0
  5377.3     .16       0  5498.2     .07       0  5658.4     .16       0
  5801.5     .07       0
Bank Sta=4994.4,5022.3
XS Rating Curve= 0 ,0
Exp/Cntr=0.3,0.1

Type RM Length L Ch R = 1 ,15383   ,599,599,599
BEGIN DESCRIPTION:
Holder Creek 22.0
END DESCRIPTION:
XS GIS Cut Line= 3
      1417454.98      6813588.01      1418256.65      6813134.01
      1418504.99      6812788.01
#Sta/Elev= 30
  4078.7 2311.37  4081.6 2311.37  4086.7 2313.95  4124.2 2305.35  4129.9 2305.58
  4136.2 2302.92  4182.2 2297.19  4232.4 2296.14  4291.6 2293.17  4313.2 2293.56
  4423.5 2285.23  4593.2 2275.37  4717.2 2272.51  4733.1 2269.25  4738.9 2266.19
  4760.5 2264.55  4848.7 2266.18  4884.6 2265.43  4916.4 2267.07  4981.3 2264.79
  5010.4 2259.74  5010.9 2259.24  5038.3 2259.74  5039.1 2265.68  5045.3 2268.03
  5139.8 2270.68  5160.7 2272.96  5175.4 2276.12  5261.4  2285.5  5425.9 2293.05
#Mann= 3 ,-1 , 0
  4078.7     .07       0  5010.4     .07       0  5038.3     .07       0
Bank Sta=5010.4,5038.3
XS Rating Curve= 0 ,0
Exp/Cntr=0.3,0.1

Type RM Length L Ch R = 1 ,14784   ,600,600,600
BEGIN DESCRIPTION:
Holder Creek 21.0
END DESCRIPTION:
XS GIS Cut Line= 3
      1417555.03      6814237.98      1418704.52       6813458.4
      1419055.02      6813187.98
#Sta/Elev= 30
  3611.1  2388.5  3618.5 2388.94  3647.3 2375.89  3654.5 2365.19  3690.4 2342.14
  3696.5 2336.07  3756.1 2305.02  3777.2 2297.34  3849.1 2284.94  4079.7 2272.18
  4259.4  2266.8  4690.7 2269.08  4741.6 2264.48  4870.4 2267.27  4951.2 2263.28
  4978.2 2258.31  4979.2 2256.25  4979.7 2255.75  5007.2 2256.25  5007.9 2258.25
  5015.2 2259.05    5064 2258.94    5093 2266.81  5102.7 2267.06  5140.3 2268.45
  5271.5 2283.56    5286  2288.6  5295.1 2288.76    5315  2294.4  5442.7 2299.29
#Mann= 7 ,-1 , 0
  3611.1     .07       0  4979.2     .07       0  5007.2     .07       0
  5015.2     .16       0  5102.7     .07       0  5140.3     .16       0
  5295.1     .07       0
#XS Ineff= 2 , 0
         4695.01 2280.08
Permanent Ineff=
       F       F
Bank Sta=4979.2,5007.2
XS Rating Curve= 0 ,0
Exp/Cntr=0.3,0.1

Type RM Length L Ch R = 1 ,14184   ,499,499,499
BEGIN DESCRIPTION:
Holder Creek 20.0
END DESCRIPTION:
XS GIS Cut Line= 3
      1417754.98      6814288.01      1418578.27      6813914.64
      1419005.04        6813888.
#Sta/Elev= 30
    4096 2303.94  4127.9 2296.69  4156.5 2287.65  4202.7 2277.68  4225.7 2275.84
  4282.9 2274.82  4346.7 2270.64    4450 2268.07  4490.7 2265.42  4858.9 2266.55
  4875.6 2265.56    4882 2262.51  4887.5 2262.51  4905.1 2257.97  4928.2 2255.35
  4933.7 2256.38  4937.2 2251.78  4937.7 2251.28  4965.4 2251.78  4974.4 2254.15
  4979.8 2252.28  5024.1 2259.41  5029.1 2258.85  5056.8 2262.83    5147 2267.53
  5184.5 2272.26  5227.2 2273.58  5287.3 2281.05  5349.9 2284.78  5427.6 2285.98
#Mann= 3 ,-1 , 0
    4096     .07       0  4937.2     .07       0  4965.4     .07       0
Bank Sta=4937.2,4965.4
XS Rating Curve= 0 ,0
Exp/Cntr=0.3,0.1

Type RM Length L Ch R = 1 ,13685   ,598,598,598
BEGIN DESCRIPTION:
Holder Creek 19.0
END DESCRIPTION:
XS GIS Cut Line= 3
      1417805.02      6814637.99      1418405.52      6814353.22
      1419004.99        6814538.
#Sta/Elev= 30
  4335.4 2397.46  4349.5 2392.84  4401.8 2348.77  4412.2 2341.91  4417.7 2335.73
  4434.9 2326.32    4446 2317.49  4457.1 2313.97  4463.2 2309.01  4479.3 2303.15
  4485.9 2298.38  4531.4 2283.52  4554.1 2278.26  4605.1 2269.55  4673.4 2264.89
  4911.8 2263.65  4944.1 2256.44  4957.3 2257.58  4995.8  2251.8  4996.3  2251.3
    5024  2251.8  5029.4  2255.6  5093.6 2258.64  5203.2 2256.45  5241.1 2258.69
  5339.1 2258.11    5513 2264.46  5578.3 2272.19  5595.9 2280.08  5627.3 2288.61
#Mann= 3 ,-1 , 0
  4335.4     .07       0  4995.8     .07       0    5024     .07       0
Bank Sta=4995.8,5024
XS Rating Curve= 0 ,0
Exp/Cntr=0.3,0.1

Type RM Length L Ch R = 1 ,13087   ,591,591,591
BEGIN DESCRIPTION:
Holder Creek 18.0
END DESCRIPTION:
XS GIS Cut Line= 3
      1417855.01        6814838.      1418644.81      6814838.55
      1419005.03      6814587.98
#Sta/Elev= 30
  4210.2 2325.36  4212.7 2325.36  4230.2 2316.16  4260.2 2306.94  4300.2 2297.08
  4340.2 2291.53  4510.2 2271.65  4660.2 2262.41  4698.1 2262.02  4760.2 2261.18
  4800.2 2252.09  4870.2 2252.23  4890.2 2250.69    4906 2247.63  4906.5 2247.13
  4934.4 2247.63  4940.2 2250.05  4950.2    2251  5004.3 2250.92  5009.4 2250.95
  5130.2 2249.93  5136.3 2253.46  5151.2 2256.35  5251.6 2256.74  5316.9  2260.8
  5365.9 2267.91  5395.6 2274.59  5402.2 2278.69  5416.5 2284.79  5438.8 2288.67
#Mann= 7 ,-1 , 0
  4210.2     .07       0  4698.1     .16       0    4906     .07       0
  4934.4     .16       0  5004.3     .07       0  5009.4     .16       0
  5251.6     .07       0
Bank Sta=4906,4934.4
XS Rating Curve= 0 ,0
Exp/Cntr=0.3,0.1

Type RM Length L Ch R = 1 ,12496   ,573,573,573
BEGIN DESCRIPTION:
Holder Creek 17.0
END DESCRIPTION:
XS GIS Cut Line= 3
      1418155.03      6815487.99      1418954.92      6815138.03
      1419555.04        6815088.
#Sta/Elev= 30
  4126.9 2290.17  4159.2 2286.62  4170.5  2282.5  4216.9 2275.58  4279.7 2269.92
  4346.7 2267.12  4650.8 2260.31  4683.2 2257.21  4694.5 2254.07  4728.2 2252.08
  4816.5 2252.03  4892.1 2249.21  4923.7 2250.53  4962.3 2247.45  4976.2 2248.13
  4991.1 2248.07  4995.6 2241.67  4996.1 2241.17  5024.7 2241.67  5030.2 2251.14
  5040.2 2254.88  5210.8 2263.59  5291.1 2264.87  5341.3 2268.42  5381.4 2280.18
  5448.9 2290.66  5491.8 2292.96  5521.9 2302.76  5595.6 2314.81  5602.2 2315.36
#Mann= 8 ,-1 , 0
  4126.9     .07       0  4346.7     .16       0  4728.2     .07       0
  4976.2     .16       0  4995.6     .07       0  5024.7     .16       0
  5448.9     .07       0  5595.6     .16       0
Bank Sta=4995.6,5024.7
XS Rating Curve= 0 ,0
Exp/Cntr=0.3,0.1

Type RM Length L Ch R = 1 ,11923   ,588,588,588
BEGIN DESCRIPTION:
Holder Creek 16.0
END DESCRIPTION:
XS GIS Cut Line= 3
      1418204.99        6815538.      1418984.61      6815668.08
      1419555.02      6815137.98
#Sta/Elev= 30
  4209.6 2288.38  4242.5 2287.12  4270.4 2278.08  4340.5 2268.88    4676 2255.58
  4817.9 2254.25  4838.2 2251.75  4850.5 2254.78  4919.3 2246.44  4980.1 2244.61
  4983.1 2240.97  4983.6 2240.47  5012.2 2240.97  5014.2  2243.3  5021.6 2244.53
  5054.5 2245.91  5170.1  2248.8  5291.2 2247.66    5326 2247.96  5389.5 2254.32
  5509.7 2261.43  5580.5 2268.77  5629.5  2277.3  5651.4  2283.5  5658.2 2282.03
  5679.7  2286.7  5700.7  2287.9  5714.9 2293.19  5736.4 2305.55  5778.7 2314.12
#Mann= 7 ,-1 , 0
  4209.6     .07       0  4340.5     .16       0  4983.1     .07       0
  5012.2     .16       0  5054.5     .07       0  5291.2     .16       0
  5629.5     .07       0
Bank Sta=4983.1,5012.2
XS Rating Curve= 0 ,0
Exp/Cntr=0.3,0.1

Type RM Length L Ch R = 1 ,11335   ,597,597,597
BEGIN DESCRIPTION:
Holder Creek 15.0
END DESCRIPTION:
XS GIS Cut Line= 3
      1417855.01        6816138.      1419451.85      6815946.32
      1419604.99      6815188.03
#Sta/Elev= 30
  3391.7 2313.17  3430.3 2311.22  3522.6 2292.31  3955.7 2266.26  4150.9 2258.76
  4368.7 2249.05  4736.6 2251.55  4821.9 2243.43  4940.8 2243.78  4952.8 2241.57
  4958.4 2236.78  4958.9 2236.28  4987.5 2236.78  5008.5 2239.33  5042.7  2248.3
  5089.9 2249.86    5156 2252.41  5189.9 2254.31  5222.7 2261.05  5232.9 2261.13
  5240.6 2258.27  5263.5 2258.99  5314.5 2266.77  5355.4 2266.41  5392.8 2262.96
  5518.6 2271.77  5620.6 2276.11    5641 2279.36  5755.4 2310.35  5773.6 2312.71
#Mann= 9 ,-1 , 0
  3391.7     .07       0  4150.9     .16       0  4736.6     .07       0
  4958.4     .07       0  4987.5     .07       0  5089.9     .16       0
    5156     .07       0  5392.8     .16       0  5755.4     .07       0
#XS Ineff= 2 , 0
         4738.69 2260.95
Permanent Ineff=
       F       F
Bank Sta=4958.4,4987.5
XS Rating Curve= 0 ,0
Exp/Cntr=0.3,0.1

Type RM Length L Ch R = 1 ,10738   ,572,572,572
BEGIN DESCRIPTION:
Holder Creek 14.0
END DESCRIPTION:
XS GIS Cut Line= 3
      1417955.01        6816388.      1419555.09      6816482.96
      1419955.03      6816588.01
#Sta/Elev= 30
  3397.1 2301.42  3456.2 2296.95  3497.3 2291.83  3646.4 2279.56  3717.7 2276.23
  3797.8 2268.76    3898 2265.06  3985.5 2258.18  4137.9 2250.84  4329.6 2245.39
    4509 2246.56  4605.1 2249.18  4689.4 2249.96  4809.6 2242.87  4909.7 2243.65
  4941.1 2240.26  4969.9 2238.64  4975.3 2233.79  4975.8 2233.29  5004.5 2233.79
  5010.2 2239.21  5041.1 2248.88  5078.2 2254.77  5199.2 2260.94  5268.7 2267.81
  5315.2 2273.38  5350.3 2281.13  5372.1 2288.52  5395.9 2291.32  5413.5  2290.6
#Mann= 8 ,-1 , 0
  3397.1    .035       0  3456.2     .07       0  4137.9     .16       0
  4605.1     .07       0  4941.1     .16       0  4975.3     .07       0
  5004.5     .16       0  5041.1     .07       0
#XS Ineff= 2 , 0
         4677.07 2265.31
Permanent Ineff=
       F       F
Bank Sta=4975.3,5004.5
XS Rating Curve= 0 ,0
Exp/Cntr=0.3,0.1

Type RM Length L Ch R = 1 ,10166   ,600,600,600
BEGIN DESCRIPTION:
Holder Creek 13.0
END DESCRIPTION:
XS GIS Cut Line= 3
      1417905.03      6816488.01       1419505.5      6817038.51
      1419954.99        6817088.
#Sta/Elev= 30
  3307.5 2305.31  3317.8 2303.08  3323.1 2306.58    3349 2302.43  3354.3  2304.1
  3360.3 2300.99  3461.8 2293.13  3707.1 2276.31  3817.6 2268.34  3848.8 2269.39
    3906 2262.36    4134 2250.08  4280.8    2244  4795.9 2246.04  4832.4  2245.3
  4872.6 2237.48  4937.6 2238.28  4967.7 2236.02  4974.2 2230.59  4974.7 2230.09
  5003.5 2230.59  5009.6 2235.36  5029.7 2239.99  5119.5 2243.23  5313.4  2251.4
  5341.5 2254.82  5391.9 2266.91  5406.7 2272.63  5432.1 2288.63  5452.2 2293.59
#Mann= 9 ,-1 , 0
  3307.5     .07       0  3461.8    .035       0  3707.1     .07       0
    4134     .16       0  4937.6     .07       0  4974.2     .07       0
  5003.5     .07       0  5119.5     .16       0  5313.4     .07       0
Bank Sta=4974.2,5003.5
XS Rating Curve= 0 ,0
Exp/Cntr=0.3,0.1

Type RM Length L Ch R = 1 ,9566    ,648,648,648
BEGIN DESCRIPTION:
Holder Creek 12.0
END DESCRIPTION:
XS GIS Cut Line= 3
      1417804.98      6816587.99      1419425.49       6817568.2
      1420004.97        6817488.
#Sta/Elev= 30
  3106.1 2324.11  3135.2 2315.65  3199.6 2305.54  3441.7 2287.21  3484.4 2287.47
  3499.9 2283.92  3506.8 2284.59  3521.3 2281.64  3581.6 2277.06  4022.1 2251.81
  4074.5 2249.89  4135.9 2247.45  4204.7 2244.25  4496.9 2242.48  4613.8 2238.34
  4817.2 2238.61  4838.5 2234.71  4906.6  2234.9  4976.3 2234.21  5009.6 2231.39
  5015.1  2229.1  5015.6  2228.6  5044.4  2229.1  5060.1  2236.2  5312.5 2237.84
  5393.2  2244.4  5423.5 2250.03  5477.3 2266.46  5524.5 2275.48    5585 2290.12
#Mann= 9 ,-1 , 0
  3106.1     .07       0  3506.8    .035       0  3581.6     .07       0
  4022.1     .16       0  4074.5     .07       0  4135.9     .16       0
  4906.6     .07       0  5015.1     .07       0  5044.4     .07       0
Bank Sta=5015.1,5044.4
XS Rating Curve= 0 ,0
Exp/Cntr=0.3,0.1

Type RM Length L Ch R = 1 ,8918    ,528,528,528
BEGIN DESCRIPTION:
Holder Creek 11.1
END DESCRIPTION:
XS GIS Cut Line= 3
      1418236.64      6818056.54       1419006.7      6818049.02
      1419888.67      6817564.48
#Sta/Elev= 30
  4229.9 2280.15  4268.3 2278.29  4348.3 2270.14  4448.3 2267.44  4508.3 2260.86
  4698.3 2250.95  4818.3 2249.62  4848.3 2243.85  4908.3 2236.15  4938.3 2226.59
  4958.3 2228.76  4978.3 2226.85  4981.4 2224.52  4981.9 2224.02  5011.8 2224.52
  5029.9 2227.64  5035.6 2225.31  5051.7 2229.83  5057.4 2226.76  5066.5 2230.32
  5123.6 2229.79  5133.2 2232.21  5138.9 2229.47    5155  2233.4  5374.6 2239.77
  5676.3 2241.21  5876.6 2241.94  5956.5 2244.62  5986.8 2248.76  6006.3 2249.37
#Mann= 4 ,-1 , 0
  4229.9     .07       0  4981.4     .07       0  5011.8     .07       0
  5676.3     .16       0
Bank Sta=4981.4,5011.8
XS Rating Curve= 0 ,0
Exp/Cntr=0.3,0.1

Type RM Length L Ch R = 1 ,8390    ,597,597,597
BEGIN DESCRIPTION:
Holder Creek 11.0
END DESCRIPTION:
XS GIS Cut Line= 3
      1418489.83      6819168.42      1419138.42      6818371.12
        1419955.        6817588.
#Sta/Elev= 30
  3972.2 2281.12  4039.8 2271.68  4111.6 2266.71  4295.4 2260.91  4509.5 2249.36
  4568.3 2249.51  4651.7 2252.26  4701.3 2251.68  4872.2 2248.55  4942.6 2242.66
  4971.3 2233.28  4985.7 2224.16  4992.1 2222.55  4998.8 2224.33  5005.8 2221.66
  5006.3 2221.16  5036.4 2221.66  5042.2 2226.82  5098.8 2230.66  5127.1  2228.8
  5162.3  2231.1  5266.8  2231.2  5335.3 2237.13  5738.1 2240.11  5896.8 2240.95
  5911.6 2241.04  5961.7 2241.34  6067.7 2246.69    6096 2252.75  6131.4 2265.09
#Mann= 10 ,-1 , 0
  3972.2     .07       0  4568.3     .16       0  4701.3     .07       0
  5005.8     .07       0  5036.4     .07       0  5266.8     .16       0
  5335.3     .07       0  5738.1     .16       0  5896.8     .07       0
  5911.6     .16       0
Bank Sta=5005.8,5036.4
XS Rating Curve= 0 ,0
Exp/Cntr=0.3,0.1

Type RM Length L Ch R = 1 ,7793    ,599,599,599
BEGIN DESCRIPTION:
Holder Creek 10.0
END DESCRIPTION:
XS GIS Cut Line= 3
      1419255.03      6818637.98      1419656.37       6818373.4
      1420055.01      6817587.98
#Sta/Elev= 30
  4519.3 2246.57  4541.9 2244.62  4555.2 2241.58  4568.9 2235.27  4591.1 2229.95
  4635.2  2231.3  4722.5 2229.92  4770.8  2226.6  4911.2 2226.37  4945.3 2225.17
  4960.4 2221.72  4974.4 2221.78  4980.9  2218.1  4981.4  2217.6  5011.5  2218.1
  5017.3  2229.2  5032.1 2234.76  5286.4 2236.17    5413 2239.72  5566.8 2244.87
    5622 2244.96  5627.6  2246.5  5634.1 2245.28  5738.9 2249.68  5769.9 2257.37
  5805.7 2266.92  5811.1 2270.46  5844.6 2285.69  5866.8 2288.21  5880.8 2285.69
#Mann= 7 ,-1 , 0
  4519.3     .07       0  4911.2     .16       0  4980.9     .07       0
  5011.5     .16       0    5413     .07       0  5769.9     .16       0
  5811.1     .07       0
Bank Sta=4980.9,5011.5
XS Rating Curve= 0 ,0
Exp/Cntr=0.3,0.1

Type RM Length L Ch R = 1 ,7194    ,568,568,568
BEGIN DESCRIPTION:
Holder Creek 9.0
END DESCRIPTION:
XS GIS Cut Line= 3
      1419154.99        6818738.      1419975.49       6818857.8
      1420504.99      6818188.01
#Sta/Elev= 30
  4170.8  2248.7  4221.3 2244.13  4302.2  2239.5  4312.3 2237.83  4345.8 2238.76
  4362.8 2234.79  4415.7 2232.93  4544.7 2233.08  4787.3 2230.35  4825.5 2226.57
  4830.6 2227.78  4878.2 2221.64  4908.5  2220.7  4928.8 2221.54    4949 2219.31
  4950.1 2218.04  4950.6 2217.54  4980.8 2218.04  5003.1 2220.53  5013.1 2224.35
  5021.1  2225.8  5056.4 2229.41  5068.8 2229.52  5178.2  2230.4  5378.6 2237.97
  5647.9 2249.04  5776.1 2263.42  5796.9 2268.79  5840.2 2274.58  5853.8 2277.89
#Mann= 5 ,-1 , 0
  4170.8     .07       0  4950.1     .07       0  4980.8     .07       0
  5068.8     .16       0  5378.6     .07       0
Bank Sta=4950.1,4980.8
XS Rating Curve= 0 ,0
Exp/Cntr=0.3,0.1
