--- Idlewild Creek.prj (project) ---

Proj Title=Idlewild Creek Base Level Engineering
Current Plan=p01
Default Exp/Contr=0.3,0.1
English Units
Geom File=g01
Flow File=f01
Plan File=p01
Y Axis Title=Elevation
X Axis Title(PF)=Main Channel Distance
X Axis Title(XS)=Station
BEGIN DESCRIPTION:
Idlewild Creek
END DESCRIPTION:
DSS Export Rating Curves= 0
DSS Export Rating Curve Sorted= 0
DSS Export Volume Flow Curves= 0
DXF OffsetX= 0
DXF OffsetY= 0
DXF ScaleX= 1
DXF ScaleY= 10

--- Idlewild Creek.p01 (plan) ---

Plan Title=Multiple Run
Short Identifier=Multiple
Geom File=g01
Flow File=f01
Subcritical Flow
K Sum by GR= 0
Std Step Tol= 0.01
Critical Tol= 0.01
Num of Std Step Trials= 20
Max Error Tol= 0.3
Flow Tol Ratio= 0.001
Split Flow NTrial= 30
Split Flow Tol= 0.02
Split Flow Ratio= 0.02
Log Output Level= 0
Friction Slope Method= 1
Unsteady Friction Slope Method= 2
Unsteady Bridges Friction Slope Method= 1
Parabolic Critical Depth
Global Vel Dist=  1 , 1 , 1
Global Log Level= 0
CheckData=True
Encroach Param= -1, 0, 0, 0
BEGIN DESCRIPTION:
Multiple Run
END DESCRIPTION:

--- Idlewild Creek.f01 (steady flow) ---

Flow Title=Multiple
Program Version=4.10
Number of Profiles= 7
Profile Names=10-year,25-year,50-year,1pct_min,100-year,1pct_plu,500-year
River Rch & RM=Idlewild Creek,Reach-1         ,27133
     183     257     319     197     394     785     608
River Rch & RM=Idlewild Creek,Reach-1         ,22162
     450     659     839     530    1058    2112    1710
River Rch & RM=Idlewild Creek,Reach-1         ,15267
     459     672     856     541    1079    2153    1742
River Rch & RM=Idlewild Creek,Reach-1         ,12337
     537     789    1008     639    1274    2543    2066
River Rch & RM=Idlewild Creek,Reach-1         ,6457
     634     932    1192     755    1507    3007    2443
Boundary for River Rch & Prof#=Idlewild Creek,Reach-1         , 1
Up Type= 0
Dn Type= 3
Dn Slope=0.021
Boundary for River Rch & Prof#=Idlewild Creek,Reach-1         , 2
Up Type= 0
Dn Type= 3
Dn Slope=0.021
Boundary for River Rch & Prof#=Idlewild Creek,Reach-1         , 3
Up Type= 0
Dn Type= 3
Dn Slope=0.021
Boundary for River Rch & Prof#=Idlewild Creek,Reach-1         , 4
Up Type= 0
Dn Type= 3
Dn Slope=0.021
Boundary for River Rch & Prof#=Idlewild Creek,Reach-1         , 5
Up Type= 0
Dn Type= 3
Dn Slope=0.021
Boundary for River Rch & Prof#=Idlewild Creek,Reach-1         , 6
Up Type= 0
Dn Type= 3
Dn Slope=0.021
Boundary for River Rch & Prof#=Idlewild Creek,Reach-1         , 7
Up Type= 0
Dn Type= 3
Dn Slope=0.021
DSS Import GetInterval= 0
DSS Import GetPeak= 0
DSS Import FillOption= 0

--- Idlewild Creek.g01 (geometry) ---

Geom Title=Existing Conditions
Program Version=4.10

River Reach=Idlewild Creek  ,Reach-1
Reach XY= 30
        1358205.        6850188.      1359182.22      6849987.71
      1360194.45      6850336.92      1360741.67      6849551.39
      1361456.43      6849241.06      1362734.74      6849488.14
      1362906.65       6849041.1      1364197.46      6848834.94
      1364158.19      6848446.35      1364741.64      6848151.34
      1364996.92       6847491.3      1364459.95      6846990.57
      1364610.85      6846790.06      1365294.56      6847036.95
       1365794.3       6846588.7      1366701.69      6846979.98
      1367007.86      6846843.08      1367170.16      6847288.48
      1367951.78      6846845.83      1368207.55      6847032.28
      1368360.84      6846640.05      1369357.74      6846732.66
      1368918.37      6846274.68      1370561.21       6845530.2
      1371051.66      6844786.28      1370805.37      6844272.83
      1370918.36      6843374.65      1371411.48      6843330.31
       1371945.2      6842548.48        1373505.        6841688.

Type RM Length L Ch R = 1 ,27133   ,582,582,582
BEGIN DESCRIPTION:
Idlewild Creek 50.0
END DESCRIPTION:
XS GIS Cut Line= 3
      1358354.99      6850288.05      1358386.81      6850137.98
        1358405.      6849987.98
#Sta/Elev= 30
  4846.6 2358.68  4856.9 2358.33  4866.4 2357.34  4871.5 2357.12  4887.5 2353.43
  4897.8 2350.52    4916 2343.65  4921.1 2342.57  4928.4 2340.51  4936.6 2340.43
  4936.9 2339.93  4940.4 2339.93  4940.6 2340.43  4959.1 2341.12  4965.7    2341
  4970.8 2340.47  4979.5 2340.69  5002.5 2340.71  5020.1 2341.02  5025.8 2340.83
  5030.9 2342.04  5040.3 2342.82  5050.4 2344.01  5060.4 2345.65  5080.6 2348.56
  5090.6 2351.26  5120.9 2357.04  5130.9 2358.01    5141 2360.54  5151.1 2360.94
#Mann= 3 ,-1 , 0
  4846.6     .07       0  4936.6     .07       0  4940.6     .07       0
Bank Sta=4936.6,4940.6
XS Rating Curve= 0 ,0
Exp/Cntr=0.3,0.1

Type RM Length L Ch R = 1 ,26551   ,490,490,490
BEGIN DESCRIPTION:
Idlewild Creek 49.0
END DESCRIPTION:
XS GIS Cut Line= 3
      1358704.97      6850438.03       1358968.9      6850138.52
      1358704.98      6849887.98
#Sta/Elev= 30
  4600.8 2362.38  4650.6 2355.32  4664.9 2354.26  4671.5 2352.28  4693.3 2349.01
  4707.5 2347.74  4714.2 2346.22  4771.1 2340.57  4799.6 2338.73  4806.2  2339.3
  4834.7 2336.32  4905.8 2332.97  4926.7 2332.37  4947.6 2333.14  4988.3 2331.51
  4988.5 2331.01  4992.3 2331.51  5017.4 2332.45  5024.3 2331.83  5123.4 2336.94
  5165.9  2341.3  5172.8 2342.73  5201.1 2344.87  5215.2 2346.94  5229.4 2350.36
  5250.8 2358.49  5279.1 2363.54  5335.7 2371.36  5360.4 2375.62  5363.9 2375.62
#Mann= 3 ,-1 , 0
  4600.8     .07       0  4988.3     .07       0  4992.3     .07       0
Bank Sta=4988.3,4992.3
XS Rating Curve= 0 ,0
Exp/Cntr=0.3,0.1

Type RM Length L Ch R = 1 ,26061   ,405,405,405
BEGIN DESCRIPTION:
Idlewild Creek 48.0
END DESCRIPTION:
XS GIS Cut Line= 3
      1359454.99      6850337.97      1359360.17      6850037.58
      1359654.98      6849738.02
#Sta/Elev= 30
    4685 2344.47  4686.3 2344.47  4687.6 2344.47  4701.1 2338.57  4706.4 2338.86
  4716.4 2337.18  4733.5 2333.14  4779.4 2332.09  4798.2 2330.54  4803.4 2330.93
  4830.5 2329.24  4835.7 2329.45  4904.2 2326.14  4965.1  2324.3  4989.1 2324.64
  4995.2 2324.17  4995.4 2323.67  4998.9 2323.67  4999.2 2324.17  5052.7 2324.85
  5158.7 2328.93  5194.1 2332.03  5229.4 2332.69  5271.8 2334.78  5328.4 2338.91
    5385 2341.88  5406.2 2343.66  5413.3 2344.47  5416.8 2345.75  5420.3 2345.75
#Mann= 5 ,-1 , 0
    4685     .07       0  4686.3    .035       0  4904.2     .07       0
  4995.2     .07       0  4999.2     .07       0
Bank Sta=4995.2,4999.2
XS Rating Curve= 0 ,0
Exp/Cntr=0.3,0.1

Type RM Length L Ch R = 1 ,25656   ,549,549,549
BEGIN DESCRIPTION:
Idlewild Creek 47.0
END DESCRIPTION:
XS GIS Cut Line= 3
      1359554.99      6850438.02       1359727.8      6850137.81
      1359854.98      6849988.02
#Sta/Elev= 30
  4653.6 2361.86  4661.5 2359.56  4667.3 2359.35  4683.1 2348.71  4714.5 2338.13
  4734.4 2333.06  4785.1 2330.78  4828.2 2326.48  4881.4 2323.18  4908.7 2317.98
  4918.7 2318.51  4924.5 2317.02  4940.3 2322.56  4946.1 2320.49  4953.6 2321.67
  4961.9 2319.95  4967.6 2315.73  4981.4 2314.51  4981.7 2314.01  4985.4 2314.51
  5012.6 2316.38    5026 2319.74  5033.4 2323.11  5068.6 2324.09    5118 2330.63
  5154.3 2336.23  5168.5 2339.34  5175.1 2342.07  5182.8  2342.2  5196.5 2345.31
#Mann= 5 ,-1 , 0
  4653.6     .07       0  4714.5    .035       0  4785.1     .07       0
  4981.4     .07       0  4985.4     .07       0
Bank Sta=4981.4,4985.4
XS Rating Curve= 0 ,0
Exp/Cntr=0.3,0.1

Type RM Length L Ch R = 1 ,25107   ,497,497,497
BEGIN DESCRIPTION:
Idlewild Creek 46.0
END DESCRIPTION:
XS GIS Cut Line= 3
      1360305.02      6850488.04      1360207.32      6850332.36
      1360004.99      6850037.99
#Sta/Elev= 30
  4816.2  2331.1  4845.1 2328.36  4851.7 2326.31  4881.6  2320.7  4887.5 2320.51
  4918.2 2316.68  4939.4 2315.87  4946.1 2313.58  4954.7 2311.81  4975.9 2310.12
  4997.6 2309.92  4997.9 2309.42  5001.4 2309.42  5001.6 2309.92  5012.1 2310.08
    5027 2312.35  5033.1 2312.33  5041.7 2314.97  5054.1 2316.36  5098.7 2315.96
  5140.7 2317.78  5206.3 2316.94  5227.3 2318.29  5242.2 2318.37  5248.2 2319.84
  5257.1 2320.55    5278 2319.57    5299 2319.85  5334.8 2323.23  5357.2  2326.6
#Mann= 3 ,-1 , 0
  4816.2     .07       0  4997.6     .07       0  5001.6     .07       0
Bank Sta=4997.6,5001.6
XS Rating Curve= 0 ,0
Exp/Cntr=0.3,0.1

Type RM Length L Ch R = 1 ,24610   ,498,498,498
BEGIN DESCRIPTION:
Idlewild Creek 45.0
END DESCRIPTION:
XS GIS Cut Line= 3
      1360654.99      6850087.99      1360578.71      6850014.82
      1360255.02      6849738.02
#Sta/Elev= 30
  4894.3 2311.58  4929.7    2309  4943.8 2306.49  4986.3 2304.44  4993.2 2303.49
  5007.1 2299.56  5019.4    2298  5019.7  2297.5  5023.4    2298  5029.1 2301.01
  5043.4  2303.6  5057.5  2302.6  5064.2 2304.64  5070.8 2302.81  5078.5 2302.05
  5092.8    2302  5099.3 2304.17    5107 2304.06  5121.3 2305.51  5127.9 2307.38
  5142.2 2308.76  5213.5 2310.82    5298 2316.07  5340.9 2321.98  5347.4  2323.7
  5369.4 2321.39  5383.7 2322.29  5397.9  2325.3  5418.8 2332.09  5425.9 2332.19
#Mann= 3 ,-1 , 0
  4894.3     .07       0  5019.4     .07       0  5023.4     .07       0
Bank Sta=5019.4,5023.4
XS Rating Curve= 0 ,0
Exp/Cntr=0.3,0.1

Type RM Length L Ch R = 1 ,24112   ,477,477,477
BEGIN DESCRIPTION:
Idlewild Creek 44.0
END DESCRIPTION:
XS GIS Cut Line= 3
      1360805.01      6849788.02      1360724.72      6849567.48
        1360705.      6849437.98
#Sta/Elev= 30
  4765.3 2304.37  4775.3 2303.89  4818.5 2303.98  4829.2  2303.6  4850.5 2303.83
    4867 2302.99  4882.4 2303.22  4897.6 2302.33  4903.7 2301.46  4914.3    2301
  4922.9 2299.86  4928.2 2300.02  4935.6 2298.82  4946.2 2297.98  4953.4 2296.75
  4978.2 2295.58  4989.3 2295.48  5002.3 2294.91  5009.6  2292.8  5017.7 2291.01
    5018 2290.51  5021.5 2290.51  5021.7 2291.01  5033.1 2292.45  5050.1 2298.93
  5060.2 2301.52  5096.7 2304.87  5101.7 2304.85  5120.9 2306.04    5131  2306.3
#Mann= 3 ,-1 , 0
  4765.3     .07       0  5017.7     .07       0  5021.7     .07       0
Bank Sta=5017.7,5021.7
XS Rating Curve= 0 ,0
Exp/Cntr=0.3,0.1

Type RM Length L Ch R = 1 ,23635   ,479,479,479
BEGIN DESCRIPTION:
Idlewild Creek 43.0
END DESCRIPTION:
XS GIS Cut Line= 3
        1361155.      6849737.99      1361160.18      6849438.44
      1361055.02      6849338.02
#Sta/Elev= 30
  4700.4 2301.35  4770.4 2297.24  4840.4 2294.51  4870.4 2291.79  4890.4 2291.58
  4920.4  2294.4  4930.4 2294.74  4940.4 2294.31  4960.4  2294.7  4970.4    2294
  4980.4 2291.38  4987.5 2290.24  4992.5 2290.16  4997.7 2287.82    5009 2287.33
  5009.2 2286.83  5012.7 2286.83    5013 2287.33  5018.2 2287.78  5025.1 2290.56
  5032.4 2290.84  5039.3 2292.49  5053.4 2293.81  5060.7  2293.5  5081.7  2295.7
  5103.1 2296.14  5117.3 2297.53  5124.2 2298.93  5131.4 2298.77  5145.4 2300.13
#Mann= 3 ,-1 , 0
  4700.4     .07       0    5009     .07       0    5013     .07       0
Bank Sta=5009,5013
XS Rating Curve= 0 ,0
Exp/Cntr=0.3,0.1

Type RM Length L Ch R = 1 ,23156   ,499,499,499
BEGIN DESCRIPTION:
Idlewild Creek 42.0
END DESCRIPTION:
XS GIS Cut Line= 3
        1361255.        6849888.      1361538.49      6849270.79
        1361505.      6849037.99
#Sta/Elev= 30
  4320.8  2311.4  4329.5 2310.37    4335 2310.93  4375.5  2306.6  4419.8 2304.17
  4432.5 2302.75  4478.4  2301.5  4495.9 2299.94  4552.9 2297.58  4639.3 2291.97
  4644.8 2292.28  4650.9 2291.26  4667.8 2290.33  4673.3 2290.86  4719.3    2288
  4765.3 2286.75  4788.2  2286.9  4816.7 2288.58  4857.2 2288.42  4937.1 2285.03
  4977.6 2284.89  4992.1  2284.1  4996.8 2280.97    4997 2280.47  5000.8 2280.97
  5003.9 2280.97  5012.9 2283.75    5023 2285.27  5064.1  2289.6  5235.2 2294.98
#Mann= 3 ,-1 , 0
  4320.8     .07       0  4996.8     .07       0  5000.8     .07       0
Bank Sta=4996.8,5000.8
XS Rating Curve= 0 ,0
Exp/Cntr=0.3,0.1

Type RM Length L Ch R = 1 ,22657   ,495,495,495
BEGIN DESCRIPTION:
Idlewild Creek 41.0
END DESCRIPTION:
XS GIS Cut Line= 3
      1361404.99      6849888.01      1361884.64      6849287.58
        1361855.      6849137.99
#Sta/Elev= 30
  4231.5 2304.09  4309.2 2299.57  4317.2  2299.9  4387.6 2296.28  4494.9 2292.79
  4666.2    2285  4693.4 2282.85  4701.4 2279.52  4715.8 2278.67  4730.2 2280.39
  4743.5 2278.88  4765.5 2278.32  4771.9 2280.52  4800.7 2281.75  4821.5 2280.57
  4928.8  2279.8  4943.2 2276.62  4957.6 2277.65    4962    2276  4962.2  2275.5
    4966    2276    4972 2277.82  4978.4 2276.55  4986.4 2279.22  4992.8 2277.64
  4996.5 2280.11  5002.3 2280.11  5009.8 2282.73  5019.4 2284.04  5152.5 2290.39
#Mann= 3 ,-1 , 0
  4231.5     .07       0    4962     .07       0    4966     .07       0
Bank Sta=4962,4966
XS Rating Curve= 0 ,0
Exp/Cntr=0.3,0.1

Type RM Length L Ch R = 1 ,22162   ,498,498,498
BEGIN DESCRIPTION:
Idlewild Creek 40.0
END DESCRIPTION:
XS GIS Cut Line= 3
      1362554.99      6849987.98      1362310.93      6849290.24
        1362305.      6848887.98
#Sta/Elev= 30
  4260.8 2297.93    4302 2294.55  4369.4 2291.96  4377.3 2289.96  4397.4 2290.62
  4462.5 2287.67  4519.3  2286.6    4788 2274.61  4832.9 2274.35  4881.1    2272
  4912.1 2271.93  4943.2 2273.43    4960  2271.1  4968.9 2268.71  4971.8 2266.48
  4972.1 2265.98  4976.7 2266.48  4981.2 2266.52  4991.8 2270.73  5003.6 2272.17
  5022.2 2277.61  5042.2 2280.61  5058.3 2280.86  5210.9 2288.51  5252.3 2290.77
  5302.3  2297.6  5331.3 2298.39  5362.3 2299.55  5380.9 2302.34  5402.3  2306.7
#Mann= 8 ,-1 , 0
  4260.8    .035       0  4397.4     .07       0  4971.8     .07       0
  4976.7     .07       0  5058.3    .035       0  5210.9     .07       0
  5331.3    .035       0  5380.9     .07       0
Bank Sta=4971.8,4976.7
XS Rating Curve= 0 ,0
Exp/Cntr=0.3,0.1

Type RM Length L Ch R = 1 ,21664   ,588,588,588
BEGIN DESCRIPTION:
Idlewild Creek 39.0
END DESCRIPTION:
XS GIS Cut Line= 3
        1362655.      6849588.02       1362675.1      6849488.33
       1362534.6      6848945.93
#Sta/Elev= 30
  4898.3 2284.21  4918.6 2282.94  4923.7 2283.24  4939.1 2281.15  4949.3 2274.08
  4959.5 2266.04    4967 2262.25  4967.3 2261.75  4971.5 2261.75  4971.9 2262.25
  4974.5 2263.08  4979.9 2262.33  4990.1 2266.23  4997.6 2267.33  5023.2 2267.45
  5058.7 2269.62    5083 2270.36  5180.5 2269.78  5215.9 2270.72  5261.7 2273.27
  5322.3 2275.26  5361.9 2276.47  5424.1 2280.18  5436.2 2280.31  5454.4 2280.73
  5500.1 2283.55  5516.8 2282.92  5535.6 2283.78  5540.7 2284.59  5560.3 2282.54
#Mann= 5 ,-1 , 0
  4898.3     .07       0    4967     .07       0  4971.9     .07       0
  5322.3    .035       0  5436.2     .07       0
Bank Sta=4967,4971.9
XS Rating Curve= 0 ,0
Exp/Cntr=0.3,0.1

Type RM Length L Ch R = 1 ,21076   ,188,188,188
BEGIN DESCRIPTION:
Idlewild Creek 38.0
END DESCRIPTION:
XS GIS Cut Line= 3
      1362737.32      6849872.95      1362874.84       6849067.4
      1362879.41      6848636.52
#Sta/Elev= 30
  4182.8  2290.9  4421.1 2285.02  4532.7  2275.5  4551.6 2271.84  4556.7 2273.14
  4563.2 2269.54    4636 2268.89  4654.5 2264.97  4671.9  2264.2  4766.1  2263.8
  4786.4 2265.54  4797.3 2269.13  4816.8 2270.13  4897.9 2265.52  4958.8 2265.95
  5019.4 2263.46    5037  2258.5  5037.3    2258  5041.9  2258.5  5059.4 2262.43
  5119.4 2267.26  5149.4  2279.5  5159.4 2281.31  5169.4 2279.17  5189.4 2278.49
  5219.4 2285.74  5259.4  2289.1  5309.4 2290.21  5389.4 2303.06  5430.9 2306.41
#Mann= 4 ,-1 , 0
  4182.8    .035       0    4636     .07       0    5037     .07       0
  5041.9     .07       0
#XS Ineff= 2 , 0
         4799.19 2276.05
Permanent Ineff=
       F       F
Bank Sta=5037,5041.9
XS Rating Curve= 0 ,0
Exp/Cntr=0.3,0.1

Type RM Length L Ch R = 1 ,20888   ,674,674,674
BEGIN DESCRIPTION:
Idlewild Creek 37.0
END DESCRIPTION:
XS GIS Cut Line= 3
      1362836.99      6850000.96      1363024.83      6849108.41
      1363078.94      6848721.18
#Sta/Elev= 30
  4087.9 2291.15  4285.1 2285.49  4298.6 2282.47  4336.2 2282.33  4348.4 2280.53
  4601.9 2270.57    4653 2265.24  4704.1 2263.47  4724.5 2260.06  4731.7 2262.44
  4736.8 2260.47  4781.5 2269.25  4786.6 2267.86  4806.3 2269.85  4867.6  2268.4
  4925.9 2264.73  4969.8 2264.63  4980.8 2257.62  4987.7 2256.21  4988.1 2255.71
  4992.7 2256.21  5020.6 2261.55  5091.3 2263.26  5101.4 2265.39    5108 2268.91
  5202.4 2271.74    5273 2284.33  5322.4 2289.62  5363.9 2299.14    5391 2304.57
#Mann= 4 ,-1 , 0
  4087.9    .035       0  4987.7    .035       0  4992.7    .035       0
  5363.9    .063       0
#XS Ineff= 2 , 0
         4776.04 2279.63
Permanent Ineff=
       F       F
Bank Sta=4987.7,4992.7
XS Rating Curve= 0 ,0
Exp/Cntr=0.3,0.1

Type RM Length L Ch R = 1 ,20214   ,489,489,489
BEGIN DESCRIPTION:
Idlewild Creek 36.0
END DESCRIPTION:
XS GIS Cut Line= 3
      1363754.97      6849287.96      1363471.48      6848955.13
      1363304.98      6848687.97
#Sta/Elev= 30
  4562.8 2303.84  4633.6 2287.59  4654.7 2279.83  4697.3 2274.12  4719.2 2268.26
  4769.2 2264.96    4834 2260.85  4881.7 2257.25  4938.9 2257.04    4974 2252.02
  4981.7 2254.93  4985.4 2251.32  4985.9 2250.82  4991.2 2251.32  5002.7 2255.96
  5008.5 2253.49  5039.2 2258.87  5064.1 2259.65  5075.8 2263.55  5081.7 2260.01
  5097.1  2265.1  5102.9 2260.59  5112.4 2262.53  5118.3 2260.07  5133.6 2265.58
  5139.5 2263.55  5154.9 2266.38  5170.2 2272.89  5249.3 2280.47  5314.8  2291.9
#Mann= 6 ,-1 , 0
  4562.8     .16       0  4769.2     .07       0    4834     .16       0
  4985.4     .07       0  4991.2     .16       0  5064.1     .07       0
#XS Ineff= 2 , 0
                         5074.11         2268.64
Permanent Ineff=
       F       F
Bank Sta=4985.4,4991.2
XS Rating Curve= 0 ,0
Exp/Cntr=0.3,0.1

Type RM Length L Ch R = 1 ,19725   ,573,573,573
BEGIN DESCRIPTION:
Idlewild Creek 35.0
END DESCRIPTION:
XS GIS Cut Line= 3
      1363905.01      6849138.02      1363794.24       6848738.7
      1363555.02      6848488.02
#Sta/Elev= 30
  4585.6 2286.58  4602.8 2281.39  4607.9 2281.53  4627.1 2276.05  4662.2 2270.12
  4676.5 2266.26  4689.4 2260.87  4710.2 2258.33  4834.7 2256.03  4896.9  2256.9
  4969.6 2255.22  5003.1 2254.15  5021.2 2251.56  5032.4 2248.38  5032.9 2247.88
  5038.2 2248.38  5049.5 2251.69  5056.4 2251.83  5063.6 2254.97  5070.5 2255.59
  5077.8 2258.67  5084.7 2258.22  5091.9 2260.85  5101.3 2260.45    5113 2260.37
  5162.7 2268.99  5212.1 2272.24  5240.4 2275.54  5304.2 2290.56  5346.5 2295.17
#Mann= 5 ,-1 , 0
  4585.6     .07       0  4662.2     .16       0  5032.4     .07       0
  5038.2     .16       0  5101.3     .07       0
Bank Sta=5032.4,5038.2
XS Rating Curve= 0 ,0
Exp/Cntr=0.3,0.1

Type RM Length L Ch R = 1 ,19152   ,426,426,426
BEGIN DESCRIPTION:
Idlewild Creek 34.0
END DESCRIPTION:
XS GIS Cut Line= 3
      1364443.24      6848929.83      1364157.73      6848731.92
      1363719.45      6848374.57
#Sta/Elev= 30
  4652.6 2287.83  4738.3 2277.93  4875.4 2265.34  4881.6 2261.24  4890.3  2261.2
  4896.3 2259.19  4911.2  2253.1  4918.2 2248.31  4926.1 2246.02  4932.1 2247.68
  4940.9 2245.98  4961.9  2247.2  4988.2 2245.71  4988.7 2245.21  4994.2 2245.71
  4997.7 2247.42    5005 2246.06    5012 2248.51  5018.5 2246.86  5026.4  2249.8
  5040.8 2251.36  5090.3 2250.46  5096.8 2248.36  5139.9 2255.06  5154.2 2255.95
  5409.8 2268.57  5467.3 2269.11  5480.9 2270.94  5523.3 2284.52  5565.5 2294.76
#Mann= 3 ,-1 , 0
  4652.6     .07       0  4988.2     .07       0  4994.2     .07       0
#XS Ineff= 2 , 0
         4967.97 2254.55 5028.12         2256.98
Permanent Ineff=
       F       F
Bank Sta=4988.2,4994.2
XS Rating Curve= 0 ,0
Exp/Cntr=0.3,0.1

Type RM Length L Ch R = 1 ,18726   ,382,382,382
BEGIN DESCRIPTION:
Idlewild Creek 33.0
END DESCRIPTION:
XS GIS Cut Line= 3
      1364788.39      6848539.02       1364246.9      6848394.29
      1363894.72      6848256.98
#Sta/Elev= 30
  4439.5 2290.64  4494.8 2287.61  4546.5 2279.67    4650 2271.84  4681.1 2268.41
  4701.8 2263.95    4736 2261.22  4753.5 2256.55  4770.9  2256.5    4776 2255.45
  4808.8 2256.27  4891.1 2252.19  4960.6 2251.47  4981.3 2248.51  4991.6 2245.77
  4995.4 2242.47  4995.9 2241.97  5001.4 2242.47  5012.6 2247.85  5017.2 2248.22
  5059.8 2249.24  5130.8 2257.14  5216.7 2262.44  5282.7 2269.87  5301.8  2270.9
  5306.4  2272.8  5327.8  2275.9  5331.6 2276.87    5337 2282.97    5378 2290.86
#Mann= 8 ,-1 , 0
  4439.5    .063       0  4808.8    .035       0  4995.4    .035       0
  5001.4    .035       0  5012.6     .07       0  5017.2    .035       0
  5306.4     .07       0  5327.8    .035       0
Bank Sta=4995.4,5001.4
XS Rating Curve= 0 ,0
Exp/Cntr=0.3,0.1

Type RM Length L Ch R = 1 ,18344   ,612,612,612
BEGIN DESCRIPTION:
Idlewild Creek 32.0
END DESCRIPTION:
XS GIS Cut Line= 3
      1364719.27      6848375.82      1364561.08      6848279.91
      1363939.95      6848121.94
#Sta/Elev= 30
    4815 2274.08  4890.2 2269.83  4939.2  2265.3    4955 2258.88  4960.8 2251.83
  4970.5  2248.5  4976.3 2243.05  4980.7 2240.98  4981.2 2240.48  4986.7 2240.98
  5024.9 2241.14    5030 2244.45  5099.1 2245.14  5106.7 2243.74  5111.9  2245.3
  5181.7 2247.12  5188.6 2247.66  5193.7 2251.08  5202.3 2251.68    5223  2249.6
  5234.7 2253.55    5315 2256.99  5434.1 2262.43  5502.2  2267.2  5542.8 2270.85
  5573.8 2276.41  5597.8 2282.54  5625.4 2293.59  5634.8 2295.51  5640.9 2298.04
#Mann= 7 ,-1 , 0
    4815    .035       0  4939.2     .07       0  4980.7     .07       0
  4986.7     .07       0    5315    .035       0  5502.2     .07       0
  5634.8    .035       0
Bank Sta=4980.7,4986.7
XS Rating Curve= 0 ,0
Exp/Cntr=0.3,0.1

Type RM Length L Ch R = 1 ,17732   ,499,499,499
BEGIN DESCRIPTION:
Idlewild Creek 31.0
END DESCRIPTION:
XS GIS Cut Line= 3
      1364979.73        6848086.      1364704.81      6847787.92
      1364024.97      6847911.61
#Sta/Elev= 30
  4594.5 2265.01  4681.4 2262.74  4688.2 2261.41  4709.8  2261.6  4730.7 2259.65
  4752.3 2259.28  4794.8  2251.9  4815.8 2249.55    4823  2249.7  4836.8  2247.7
    4851  2248.2  4943.4 2243.71  4971.7    2241  4978.5 2239.33  4985.9 2239.63
  4993.5 2237.69    4994 2237.19  4999.6 2237.69    5010 2238.79  5020.1 2242.24
  5026.8 2246.27  5050.6 2251.18  5088.4 2252.55  5138.6 2253.84  5162.4 2255.78
  5213.3 2255.16  5367.2 2257.35  5487.7 2260.88  5613.5 2266.89    5691  2271.9
#Mann= 5 ,-1 , 0
  4594.5     .07       0  4993.5     .07       0  4999.6     .07       0
  5088.4    .035       0  5613.5     .07       0
Bank Sta=4993.5,4999.6
XS Rating Curve= 0 ,0
Exp/Cntr=0.3,0.1

Type RM Length L Ch R = 1 ,17233   ,996,996,996
BEGIN DESCRIPTION:
Idlewild Creek 30.0
END DESCRIPTION:
XS GIS Cut Line= 3
      1365055.01      6847638.01      1364985.23      6847507.83
      1364205.04      6847188.01
#Sta/Elev= 30
  4852.3 2258.91  4882.4 2257.07    4910 2251.68  4920.4 2251.97  4936.9 2245.49
  4948.2 2241.28  4964.4 2241.09  4970.1 2238.27  4986.3 2239.11    4992 2235.23
  5006.1 2235.07  5006.6 2234.57  5012.2 2235.07  5038.6 2240.06    5092 2241.48
  5110.9 2243.84  5324.1 2244.94  5382.9 2235.24  5400.1 2235.21  5465.7  2244.5
  5596.4 2251.59  5644.4 2257.24  5673.8 2258.51  5745.8 2267.57  5751.2 2266.75
  5756.8 2269.73  5804.6 2281.41  5810.8 2285.39  5828.5  2291.3  5843.2 2292.26
#Mann= 5 ,-1 , 0
  4852.3     .07       0  4936.9     .16       0  5006.1     .07       0
  5012.2     .16       0  5110.9     .07       0
Bank Sta=5006.1,5012.2
XS Rating Curve= 0 ,0
Exp/Cntr=0.3,0.1

Type RM Length L Ch R = 1 ,16237   ,476,476,476
BEGIN DESCRIPTION:
Idlewild Creek 29.0
END DESCRIPTION:
XS GIS Cut Line= 3
      1365204.99      6847337.99      1364528.24      6846864.59
      1364235.79      6846936.26
#Sta/Elev= 30
  4174.1  2253.9  4210.7 2255.77  4324.5 2250.21  4467.5 2245.59  4476.2 2243.37
  4514.8 2244.67  4568.7 2243.14  4698.9 2243.81  4777.1 2240.49  4893.1 2238.84
  4942.9 2235.05  4986.8 2235.13  5033.9 2233.29  5034.4 2232.79  5040.9 2233.29
  5065.1 2237.55  5073.8 2242.19    5079  2239.6    5096    2251  5106.3 2260.36
  5115.4 2264.13  5120.5 2262.89  5147.5 2269.04  5196.9 2274.21  5216.5 2276.92
  5245.3 2282.12  5250.5 2279.64  5281.3 2282.46  5286.9 2284.77  5301.1 2286.94
#Mann= 7 ,-1 , 0
  4174.1     .07       0  4514.8     .16       0  4986.8     .07       0
  5033.9     .07       0  5040.9     .07       0  5196.9    .035       0
  5216.5     .07       0
Bank Sta=5033.9,5040.9
XS Rating Curve= 0 ,0
Exp/Cntr=0.3,0.1

Type RM Length L Ch R = 1 ,15761   ,494,494,494
BEGIN DESCRIPTION:
Idlewild Creek 28.0
END DESCRIPTION:
XS GIS Cut Line= 3
      1365054.99      6847187.97      1364975.26      6846787.54
      1364785.99      6846244.68
#Sta/Elev= 30
  4591.7 2247.63  4612.1 2245.83  4617.2 2246.43  4652.9 2242.64  4673.4 2237.42
  4703.8 2234.83  4719.4 2231.92  4724.5 2234.02  4732.5 2232.82    4765 2229.89
  4805.8 2229.51  4897.6 2231.53  4907.8 2230.69    4980 2231.47  5002.4 2230.04
  5010.1 2225.95  5017.4  2225.8  5017.9  2225.3  5024.5  2225.8  5031.3 2230.61
  5077.8 2237.06  5084.2 2240.21  5094.8 2240.22  5103.6 2243.22  5108.9 2243.39
    5116 2246.91  5126.6 2249.49  5178.1 2252.94    5290 2258.33  5574.9 2277.58
#Mann= 5 ,-1 , 0
  4591.7     .07       0  4732.5     .16       0  5017.4     .07       0
  5024.5     .16       0  5178.1     .07       0
Bank Sta=5017.4,5024.5
XS Rating Curve= 0 ,0
Exp/Cntr=0.3,0.1

Type RM Length L Ch R = 1 ,15267   ,474,474,474
BEGIN DESCRIPTION:
Idlewild Creek 27.0
END DESCRIPTION:
XS GIS Cut Line= 3
        1365205.        6847138.       1365260.2      6847038.48
      1365154.99      6846787.97
#Sta/Elev= 30
  4886.2 2247.99  4909.1 2247.16    4916 2246.24  4953.7 2244.88  4966.2 2239.19
  4975.5 2231.64  4981.2 2231.25  4997.2 2223.28  5007.8  2222.8  5008.3  2222.3
  5014.4  2222.3  5014.9  2222.8  5021.6 2224.85  5033.1 2226.95  5039.5 2227.31
  5050.7 2228.25  5056.2  2228.2  5065.6 2229.36  5098.1 2230.58  5103.7 2231.75
  5109.1 2232.32  5208.9 2237.38  5227.9 2237.42  5233.3 2235.71  5239.1  2236.5
    5250 2239.49  5257.1 2240.04  5262.5 2239.91    5269 2241.12  5271.7 2241.12
#Mann= 5 ,-1 , 0
  4886.2     .07       0  5007.8     .07       0  5014.9     .07       0
  5039.5     .16       0  5208.9     .07       0
Bank Sta=5007.8,5014.9
XS Rating Curve= 0 ,0
Exp/Cntr=0.3,0.1

Type RM Length L Ch R = 1 ,14793   ,490,490,490
BEGIN DESCRIPTION:
Idlewild Creek 26.0
END DESCRIPTION:
XS GIS Cut Line= 3
      1365654.99      6846887.98      1365605.87      6846753.36
      1365455.02      6846638.01
#Sta/Elev= 30
  4856.7 2239.53  4866.6 2238.32  4882.7 2237.98  4902.5 2236.71  4927.7 2233.92
  4933.1    2232  4941.8 2230.74  4952.5  2231.2  4958.3 2229.56  4963.6    2227
  4983.5 2225.36  4988.8 2223.97    5000 2223.59    5004 2221.36  5008.6 2220.15
  5009.1 2219.65  5015.8 2220.15  5026.3  2220.5    5033 2222.65  5047.6 2223.08
  5053.9 2225.21  5062.1 2224.71  5076.6 2226.82  5097.4 2227.75  5118.3 2230.61
  5132.8 2233.48  5147.3 2234.68  5153.6 2236.46  5161.8 2236.28  5189.9 2239.35
#Mann= 4 ,-1 , 0
  4856.7    .035       0  4882.7     .07       0  5008.6     .07       0
  5015.8     .07       0
Bank Sta=5008.6,5015.8
XS Rating Curve= 0 ,0
Exp/Cntr=0.3,0.1

Type RM Length L Ch R = 1 ,14303   ,492,492,492
BEGIN DESCRIPTION:
Idlewild Creek 25.0
END DESCRIPTION:
XS GIS Cut Line= 3
      1365904.98      6846888.04      1365989.94      6846688.14
      1365805.01      6846288.01
#Sta/Elev= 30
  4782.8 2238.11  4913.2 2233.68  4926.5 2231.25  4950.1 2228.94  4960.1 2225.51
  4967.6 2221.71  4973.8 2217.47  4979.2 2215.16  4985.7 2215.13  4986.2 2214.63
  4992.9 2215.13  4997.4 2219.81  5002.8 2219.81  5011.2    2222  5033.2 2221.65
  5043.1 2222.75  5071.6 2222.85  5088.3 2223.89  5094.5 2226.45    5100 2224.86
    5104  2226.1  5110.3 2228.06  5117.4 2232.55  5122.9 2230.26  5154.4 2235.99
  5186.2 2239.09  5191.7 2238.83  5328.1 2248.95  5403.7 2255.63  5440.8 2260.67
#Mann= 6 ,-1 , 0
  4782.8     .07       0  4960.1     .16       0  4985.7     .07       0
  4992.9     .16       0    5104     .07       0  5328.1    .035       0
Bank Sta=4985.7,4992.9
XS Rating Curve= 0 ,0
Exp/Cntr=0.3,0.1

Type RM Length L Ch R = 1 ,13811   ,499,499,499
BEGIN DESCRIPTION:
Idlewild Creek 24.0
END DESCRIPTION:
XS GIS Cut Line= 3
        1366205.        6847088.      1366444.57      6846789.05
        1366455.      6846687.99
#Sta/Elev= 30
  4616.9 2237.79  4694.5 2234.06  4731.3 2231.02  4737.7 2231.84    4773 2226.61
    4780 2226.94  4801.8  2225.7    4901 2225.07  4929.8 2221.65  4937.3  2222.5
  4944.2 2222.05  4958.6 2219.11    4965 2219.08  4969.4 2211.25  4969.9 2210.75
  4976.2 2210.75  4976.7 2211.25  4979.4 2212.24  4987.4 2217.58  4993.8 2218.23
  4997.5 2220.58    5003 2220.58  5021.2 2227.53  5041.3 2233.92  5049.6 2237.82
  5054.6 2239.14  5061.4 2242.46  5071.4    2246    5088 2247.68  5101.6 2248.36
#Mann= 5 ,-1 , 0
  4616.9     .07       0    4780     .16       0  4969.4     .07       0
  4976.7     .16       0    5088     .07       0
Bank Sta=4969.4,4976.7
XS Rating Curve= 0 ,0
Exp/Cntr=0.3,0.1

Type RM Length L Ch R = 1 ,13312   ,498,498,498
BEGIN DESCRIPTION:
Idlewild Creek 23.0
END DESCRIPTION:
XS GIS Cut Line= 3
        1366805.      6847038.01      1366845.45      6846899.08
        1366755.      6846488.02
#Sta/Elev= 30
  4855.3 2225.06  4866.1 2224.19  4872.1 2223.18    4897 2222.76  4917.8 2221.16
  4938.6  2218.1  4944.3 2216.21  4949.5 2217.45  4969.9 2214.63  4977.8 2211.47
    4983 2213.81  4990.7  2211.3  4994.3 2209.36  4994.8 2208.86  5001.6 2209.36
  5003.1 2209.36  5011.3 2213.85  5020.9 2216.75    5026 2216.99  5031.8 2216.36
  5144.5  2219.9  5185.4 2219.77  5260.1 2221.72  5313.6 2222.28  5328.8 2223.52
  5347.6 2223.77  5369.7 2226.91    5380 2229.57  5410.7 2240.52  5420.9 2242.37
#Mann= 5 ,-1 , 0
  4855.3     .07       0  4866.1     .16       0  4994.3     .07       0
  5001.6     .16       0  5313.6     .07       0
Bank Sta=4994.3,5001.6
XS Rating Curve= 0 ,0
Exp/Cntr=0.3,0.1

Type RM Length L Ch R = 1 ,12814   ,477,477,477
BEGIN DESCRIPTION:
Idlewild Creek 22.0
END DESCRIPTION:
XS GIS Cut Line= 3
      1366739.19      6847230.79      1366954.59        6847113.
      1367304.97      6846888.02
#Sta/Elev= 30
  4754.5 2229.85  4834.2 2229.95  4886.5 2228.25  4915.8 2226.78  4921.5  2225.3
  4931.9 2224.64  4937.6 2225.11  4953.8  2218.8  4981.3 2215.39  4989.1 2212.65
  4999.5 2207.58    5000 2207.08  5006.9 2207.58  5012.4 2211.87  5043.2 2214.19
  5054.7 2214.92  5069.9 2213.97  5091.1 2214.29  5140.5 2217.56  5148.6 2217.83
  5169.7 2222.43  5184.9 2222.82  5214.4 2225.94  5236.4 2226.69  5263.5 2226.39
  5321.4 2222.46  5345.1    2223  5380.8 2230.58  5387.7 2233.23  5416.4 2238.12
#Mann= 5 ,-1 , 0
  4754.5     .07       0  4999.5     .07       0  5006.9     .07       0
  5043.2     .16       0  5140.5     .07       0
Bank Sta=4999.5,5006.9
XS Rating Curve= 0 ,0
Exp/Cntr=0.3,0.1

Type RM Length L Ch R = 1 ,12337   ,594,594,594
BEGIN DESCRIPTION:
Idlewild Creek 21.0
END DESCRIPTION:
XS GIS Cut Line= 3
      1367211.39      6847512.95      1367303.28      6847233.78
        1367355.      6846888.03
#Sta/Elev= 30
  4706.1 2230.28  4735.6 2228.01  4774.5 2228.01  4799.2 2224.48  4825.7 2226.62
    4831 2224.01  4837.6  2223.6  4857.5 2224.47  4862.8 2223.18  4885.4 2222.96
  4911.3  2221.7  4926.3 2217.04  4932.4 2212.91  4974.5 2209.92  4985.9 2205.62
  4986.4 2205.12    4994 2205.62  4995.1 2207.15    5000 2207.15  5005.8 2211.54
  5036.2 2209.36  5056.4 2212.66  5067.5 2212.86  5117.6 2212.86  5163.5 2216.16
  5250.9 2217.56  5278.8  2219.9  5309.2 2229.14    5315 2232.32  5349.6 2240.25
#Mann= 6 ,-1 , 0
  4706.1    .035       0  4885.4     .07       0  4985.9     .07       0
    4994     .07       0  5067.5     .16       0  5163.5     .07       0
Bank Sta=4985.9,4994
XS Rating Curve= 0 ,0
Exp/Cntr=0.3,0.1

Type RM Length L Ch R = 1 ,11743   ,159,159,159
BEGIN DESCRIPTION:
Idlewild Creek 20.0
END DESCRIPTION:
XS GIS Cut Line= 3
      1367661.58       6847425.4      1367704.49      6846937.49
      1367837.73      6846154.64
#Sta/Elev= 30
  4510.2 2225.88  4529.1 2224.88  4604.7 2219.58  4609.7  2220.9  4678.2 2216.08
  4725.2  2214.2  4909.1 2207.98  4921.4 2208.59  4969.4 2207.49  4985.4 2203.19
  4985.9 2202.69  4993.5 2203.19  4997.2 2205.18  5002.3 2205.18  5009.6 2207.69
  5028.9 2209.06  5131.3 2211.39  5149.3 2215.99  5154.4 2212.71  5161.8  2216.2
  5182.1 2220.71  5217.3 2221.86  5324.1 2226.28  5335.1 2225.47  5384.9 2227.68
  5450.5 2227.91  5510.7 2232.62  5585.6 2234.45    5669 2236.73  5794.1  2242.5
#Mann= 8 ,-1 , 0
  4510.2    .063       0  4529.1    .035       0  4725.2     .16       0
  4921.4     .07       0  4985.4     .07       0  4993.5     .07       0
  5217.3    .035       0  5585.6     .07       0
Bank Sta=4985.4,4993.5
XS Rating Curve= 0 ,0
Exp/Cntr=0.3,0.1

Type RM Length L Ch R = 1 ,11584   ,643,643,643
BEGIN DESCRIPTION:
Idlewild Creek 19.0
END DESCRIPTION:
XS GIS Cut Line= 3
      1367753.23      6847458.33      1367849.09      6846896.45
      1367960.92      6846312.36
#Sta/Elev= 30
    4430  2231.5  4440.5 2232.31  4479.8 2228.14  4511.5 2224.83  4703.6 2215.98
  4708.7 2216.63  4734.7 2213.56  4785.4 2210.71    4829 2209.74  4884.1 2211.32
  4889.2 2209.87  4907.1 2210.78  4944.3  2203.3  4949.4 2205.55  4984.2 2202.36
  4984.7 2201.86  4992.4 2202.36    5000 2203.54  5004.2 2205.77  5009.3 2202.47
    5029 2207.43  5069.7 2209.31  5120.6 2218.22  5172.4 2217.99  5293.7 2220.04
  5334.4 2223.83  5430.7 2228.31  5482.7  2232.4  5575.1 2235.34  5594.7 2236.07
#Mann= 6 ,-1 , 0
    4430    .063       0  4479.8    .035       0  4984.2    .035       0
  4992.4    .035       0  5172.4    .063       0  5575.1    .035       0
Bank Sta=4984.2,4992.4
XS Rating Curve= 0 ,0
Exp/Cntr=0.3,0.1

Type RM Length L Ch R = 1 ,10941   ,596,596,596
BEGIN DESCRIPTION:
Idlewild Creek 18.0
END DESCRIPTION:
XS GIS Cut Line= 3
        1368155.      6847338.02      1368235.38      6847008.48
        1368155.      6846688.01
#Sta/Elev= 30
  4660.8 2221.82  4794.6 2214.94  4835.8 2214.39  4856.4  2211.5    4877 2211.56
  4892.7 2207.85  4897.8 2209.79  4918.1 2207.49  4934.3 2203.24  4939.5 2205.52
    4949 2203.56  4969.6 2202.31    4976 2199.81  4981.2 2201.06  4993.5 2197.73
    4994 2197.23  5001.8 2197.73  5024.2 2203.72  5089.8 2205.03  5183.7 2204.29
  5188.9 2205.26  5206.7 2203.34  5224.9 2203.24  5230.1 2205.33  5247.9 2206.14
  5268.2 2213.15  5271.2 2215.06  5289.2 2217.63  5312.4 2219.97  5330.4 2220.17
#Mann= 5 ,-1 , 0
  4660.8     .07       0  4993.5     .07       0  5001.8     .07       0
  5089.8     .16       0  5268.2     .07       0
Bank Sta=4993.5,5001.8
XS Rating Curve= 0 ,0
Exp/Cntr=0.3,0.1

Type RM Length L Ch R = 1 ,10345   ,479,479,479
BEGIN DESCRIPTION:
Idlewild Creek 17.0
END DESCRIPTION:
XS GIS Cut Line= 3
        1368405.      6847088.01        1368505.      6846637.98
        1368455.      6846537.99
#Sta/Elev= 30
    4539 2216.17    4612 2215.94    4621 2215.07  4662.8 2213.89  4672.5 2213.36
  4742.6 2210.51  4846.3 2203.68  4888.6  2202.3  4948.8 2202.58    4959  2201.5
  4975.7 2200.83  4989.7 2200.48  5002.8 2200.89  5008.4 2199.11    5014 2199.91
  5018.2 2195.41  5018.7 2194.91    5026 2194.91  5026.5 2195.41  5030.7 2199.13
  5036.3 2197.91  5044.7 2203.88  5053.1  2206.2  5058.7 2206.54  5067.1 2210.28
  5075.5 2217.05    5081 2216.71  5089.4 2225.55  5097.8 2231.23  5111.8    2232
#Mann= 5 ,-1 , 0
    4539     .07       0  4662.8    .035       0  4672.5     .07       0
  5018.2     .07       0  5026.5     .07       0
Bank Sta=5018.2,5026.5
XS Rating Curve= 0 ,0
Exp/Cntr=0.3,0.1

Type RM Length L Ch R = 1 ,9866    ,474,474,474
BEGIN DESCRIPTION:
Idlewild Creek 16.0
END DESCRIPTION:
XS GIS Cut Line= 3
        1368655.        6847038.      1368878.13      6846861.99
      1368805.01      6846638.02
#Sta/Elev= 30
  4715.8 2212.31  4845.3 2209.62    4901 2209.01  4915.4 2208.01  4921.8 2205.68
  4929.9 2207.28  4936.2 2204.59  4944.3  2205.1  4950.7 2202.05  4965.1 2201.13
  4971.5 2198.42  4985.9 2196.86    4994 2195.09    4995 2193.18  4995.5 2192.68
  5003.3 2193.18  5004.7 2193.18  5014.7 2198.61    5055 2198.06  5066.2 2198.68
    5124 2198.97  5150.6 2200.43  5155.9 2201.22    5162 2203.24  5182.5 2211.46
  5186.2 2211.61  5187.8 2211.68  5193.5 2215.18  5214.4 2215.74  5235.6 2214.87
#Mann= 6 ,-1 , 0
  4715.8    .035       0  4845.3     .07       0    4995     .07       0
  5003.3     .07       0  5066.2     .16       0  5186.2     .07       0
Bank Sta=4995,5003.3
XS Rating Curve= 0 ,0
Exp/Cntr=0.3,0.1

Type RM Length L Ch R = 1 ,9392    ,1443,1443,1443
BEGIN DESCRIPTION:
Idlewild Creek 15.0
END DESCRIPTION:
XS GIS Cut Line= 3
      1369312.78      6847117.35      1369260.04       6846738.1
      1368748.41      6846525.87
#Sta/Elev= 30
  4617.1 2213.17  4675.3 2210.87  4711.1 2210.18  4838.6 2202.81    4889  2195.2
  4931.1 2192.87  4956.2 2192.94  4969.8 2193.79  4979.9 2192.25    5000 2195.05
  5012.1 2191.46  5017.5 2193.75  5031.4  2191.2  5031.9  2190.7  5040.5  2191.2
  5041.4 2195.34  5065.3  2195.1  5070.7 2196.85  5178.7 2199.96  5189.5 2199.19
  5243.2 2202.25  5272.5 2201.87  5277.9 2200.69  5306.1 2203.31  5325.7 2204.17
    5355 2202.56  5378.8 2203.09    5432  2211.8  5485.2 2212.58  5553.9 2215.97
#Mann= 6 ,-1 , 0
  4617.1    .035       0  4675.3     .07       0  4956.2     .16       0
  5031.4     .07       0  5040.5     .16       0  5306.1     .07       0
Bank Sta=5031.4,5040.5
XS Rating Curve= 0 ,0
Exp/Cntr=0.3,0.1

Type RM Length L Ch R = 1 ,7949    ,499,499,499
BEGIN DESCRIPTION:
Idlewild Creek 14.0
END DESCRIPTION:
XS GIS Cut Line= 3
       1369687.1      6846871.43      1369188.48      6846054.59
      1368744.93      6845794.46
#Sta/Elev= 30
    4043 2210.06  4182.4 2207.39  4308.4 2200.25  4397.4 2198.61  4635.5  2204.3
  4730.4    2201  4877.5 2190.92  4962.7 2191.11    4989 2186.33  4989.5 2185.83
  4998.2 2186.33  5006.5 2190.75  5022.2 2191.74    5028  2195.4  5037.8 2196.28
  5043.6 2199.97  5055.7 2197.62  5059.3 2196.75  5065.1 2200.83  5073.6 2197.67
  5080.8 2200.71  5086.6 2199.49  5116.2 2210.89  5145.2 2220.55  5176.6 2224.74
  5225.3 2226.09  5262.5 2225.77  5270.7 2224.09  5305.4 2228.48  5514.2  2233.3
#Mann= 6 ,-1 , 0
    4043    .035       0  4182.4     .07       0    4989     .07       0
  4998.2     .07       0  5055.7     .16       0  5116.2     .07       0
Bank Sta=4989,4998.2
XS Rating Curve= 0 ,0
Exp/Cntr=0.3,0.1

Type RM Length L Ch R = 1 ,7450    ,498,498,498
BEGIN DESCRIPTION:
Idlewild Creek 13.0
END DESCRIPTION:
XS GIS Cut Line= 3
      1370354.99      6846687.99      1369537.78      6845904.24
        1369555.      6845788.01
#Sta/Elev= 30
  3867.7 2218.29  3911.6  2216.2  4082.3 2207.59  4292.1 2198.95  4334.5 2190.05
  4355.6 2188.05  4391.1 2187.27  4405.3 2189.84  4433.6 2190.77  4440.5 2189.38
  4490.2 2190.36  4511.3 2187.56  4532.7 2190.62  4574.8  2189.8  4751.9 2194.13
  4857.8 2190.85  4900.3 2191.29  4921.4 2187.28  4956.9 2188.05  4973.3 2185.88
  4973.8 2185.38  4982.6 2185.88  5006.3 2192.86  5013.3 2196.66  5018.3 2195.73
  5036.6 2207.05  5046.7 2210.93  5077.1 2214.26  5087.8 2217.18  5117.5 2217.99
#Mann= 5 ,-1 , 0
  3867.7     .07       0  3911.6    .035       0  4082.3     .07       0
  4973.3     .07       0  4982.6     .07       0
#XS Ineff= 2 , 0
          4813.4 2199.69
Permanent Ineff=
       F       F
Bank Sta=4973.3,4982.6
XS Rating Curve= 0 ,0
Exp/Cntr=0.3,0.1

Type RM Length L Ch R = 1 ,6952    ,495,495,495
BEGIN DESCRIPTION:
Idlewild Creek 12.0
END DESCRIPTION:
XS GIS Cut Line= 3
      1370355.03      6846238.03      1370006.08      6845853.85
      1369754.99      6845537.99
#Sta/Elev= 30
    4481 2203.64  4558.6 2199.58  4565.8 2196.74  4573.3 2191.56    4580 2184.54
  4587.5  2183.9  4665.2 2183.78  4771.3 2187.18  4794.1 2180.65  4806.4  2177.4
  4823.3 2176.12  4823.8 2175.62  4832.8 2176.12  4863.2 2177.43  4891.6 2183.11
    4899 2186.22  4929.3 2183.44  4955.1 2181.19  5011.8  2183.7    5033 2186.29
  5055.1 2191.31  5090.3 2192.78  5111.1 2198.33    5140  2197.9  5282.5  2204.9
  5325.8 2205.52  5375.5 2213.04  5381.9 2216.05  5396.3 2218.75  5403.5  2218.3
#Mann= 6 ,-1 , 0
    4481     .07       0  4558.6    .035       0  4794.1     .07       0
  4823.3    .035       0  4832.8     .07       0  4929.3    .035       0
Bank Sta=4823.3,4832.8
XS Rating Curve= 0 ,0
Exp/Cntr=0.3,0.1

Type RM Length L Ch R = 1 ,6457    ,472,472,472
BEGIN DESCRIPTION:
Idlewild Creek 11.0
END DESCRIPTION:
XS GIS Cut Line= 3
      1370405.01      6845738.01      1370309.97      6845537.94
      1370205.02      6845388.02
#Sta/Elev= 30
  4778.5 2191.86  4787.1 2191.63  4792.6  2188.9  4798.6 2187.12  4815.4 2184.23
  4867.1 2182.68  4900.3  2180.4  4906.3  2178.9  4951.7 2177.91  4957.2  2178.5
  4974.4 2178.28  4997.1  2176.9  5017.8 2175.81  5019.5 2173.76    5020 2173.26
  5028.6 2173.26  5029.1 2173.76  5032.6 2175.09  5038.7 2175.61  5047.5 2179.12
  5053.6 2179.91    5061 2184.99  5068.4 2188.27  5104.1 2189.03  5110.2 2188.21
  5118.9 2189.37    5125 2188.51  5133.8 2190.05  5146.4 2191.11    5183 2191.94
#Mann= 5 ,-1 , 0
  4778.5    .035       0  4798.6     .16       0  4997.1     .07       0
  5019.5     .07       0  5029.1     .07       0
Bank Sta=5019.5,5029.1
XS Rating Curve= 0 ,0
Exp/Cntr=0.3,0.1

Type RM Length L Ch R = 1 ,5985    ,553,553,553
BEGIN DESCRIPTION:
Idlewild Creek 10.0
END DESCRIPTION:
XS GIS Cut Line= 3
      1370754.98      6845437.98      1370684.69       6845357.7
      1370405.05      6845288.01
#Sta/Elev= 30
  4893.3  2195.2    4894  2195.2  4914.6 2194.29  4921.3 2193.54  4928.9 2193.45
  4935.5 2192.75  4943.1 2189.98  4949.7 2185.27  4957.3 2178.91    4964 2175.09
  4971.6 2172.89  4973.4 2169.32  4973.9 2168.82  4982.5 2168.82    4983 2169.32
  4992.5 2171.77  4996.5 2174.76    5010 2175.16  5017.3 2174.63  5030.6 2175.48
  5051.2 2175.79  5071.8  2178.3  5123.4 2182.42  5146.3 2183.82  5164.6 2185.58
  5174.9 2185.52  5195.5 2186.97  5205.8 2186.93    5265  2189.7  5288.2 2189.88
#Mann= 4 ,-1 , 0
  4893.3    .035       0    4894     .07       0  4973.4     .07       0
    4983     .07       0
Bank Sta=4973.4,4983
XS Rating Curve= 0 ,0
Exp/Cntr=0.3,0.1

Type RM Length L Ch R = 1 ,5432    ,181,181,181
BEGIN DESCRIPTION:
Idlewild Creek 9.0
END DESCRIPTION:
XS GIS Cut Line= 3
      1371191.68      6845032.91      1370961.18      6844936.12
      1370668.75      6844955.92
#Sta/Elev= 30
    4750 2210.75  4757.2 2208.43  4789.8 2204.06  4803.7 2201.12  4811.5 2198.39
  4822.1 2196.97  4833.2 2193.91  4865.7 2190.22  4887.4  2190.3  4904.2 2189.37
  4919.9 2184.84  4933.4 2172.59  4943.4 2169.21  4951.7  2167.1  4957.1 2167.12
  4963.3 2165.73    4976 2165.49  4976.5 2164.99  4985.9 2165.49  5026.2 2165.79
  5036.3 2167.63  5046.3    2171  5056.3 2176.49  5066.3 2178.39  5086.4 2178.59
  5101.6 2180.01  5106.7 2179.29  5186.6  2184.8  5216.7  2186.2  5293.1 2186.88
#Mann= 4 ,-1 , 0
    4750    .035       0  4943.4     .07       0    4976     .07       0
  4985.9     .07       0
Bank Sta=4976,4985.9
XS Rating Curve= 0 ,0
Exp/Cntr=0.3,0.1

Type RM Length L Ch R = 1 ,5251    ,261,261,261
BEGIN DESCRIPTION:
Idlewild Creek 8.1
END DESCRIPTION:
XS GIS Cut Line= 3
      1371328.82      6844826.05      1371051.66      6844786.28
      1370781.86      6844787.66
#Sta/Elev= 30
    4720 2203.05  4740.3 2199.58  4745.3 2200.29  4764.3 2195.29  4784.5 2185.94
  4804.7 2181.09  4815.9 2183.86  4824.9 2183.42  4865.3 2177.62  4875.4 2176.66
  4881.4  2177.7  4886.4 2175.93  4895.6 2175.65  4905.7 2175.66  4925.9 2179.59
    4936  2180.1  4948.4 2174.82  4951.9  2172.2    4957  2171.8  4986.5 2172.17
  5011.7 2170.08  5012.2 2169.58  5021.6 2170.08  5036.7 2171.98  5116.7  2170.5
  5136.7 2171.63  5166.7 2171.17  5176.7 2177.06  5186.7 2178.89  5269.8 2183.54
#Mann= 4 ,-1 , 0
    4720    .035       0  4948.4     .07       0  5011.7     .07       0
  5021.6     .07       0
#XS Ineff= 2 , 0
         4929.64 2185.58
Permanent Ineff=
       F       F
Bank Sta=5011.7,5021.6
XS Rating Curve= 0 ,0
Exp/Cntr=0.3,0.1

Type RM Length L Ch R = 1 ,4990    ,462,462,462
BEGIN DESCRIPTION:
Idlewild Creek 8.0
END DESCRIPTION:
XS GIS Cut Line= 3
      1371105.03        6844588.      1370934.58      6844568.17
      1370654.98        6844588.
#Sta/Elev= 30
  4828.4 2184.14  4848.6 2184.49  4858.6  2181.2  4867.7 2175.73  4872.7 2177.53
  4878.8 2174.58  4888.7 2173.86  4898.9 2171.12  4929.1 2168.59  4939.2 2168.69
  4956.3 2170.34  4969.4 2170.71  4979.4 2170.18  4989.5 2167.06  4992.3 2166.69
  4992.8 2166.19  5001.8 2166.19  5002.3 2166.69  5009.6 2166.82  5039.7 2174.03
  5066.5 2176.52  5071.5 2176.42  5119.9 2179.51  5139.9 2180.11    5150 2181.77
    5160 2181.26    5180 2181.75  5207.3 2183.27  5250.2 2184.47  5280.3 2186.11
#Mann= 4 ,-1 , 0
  4828.4     .07       0  4888.7     .16       0  4992.3     .07       0
  5002.3     .07       0
Bank Sta=4992.3,5002.3
XS Rating Curve= 0 ,0
Exp/Cntr=0.3,0.1

Type RM Length L Ch R = 1 ,4528    ,498,498,498
BEGIN DESCRIPTION:
Idlewild Creek 7.0
END DESCRIPTION:
XS GIS Cut Line= 3
      1371205.02      6844388.01      1370805.51      6844153.22
      1370654.97      6844188.01
#Sta/Elev= 30
  4536.6 2189.25  4624.5 2184.35  4661.7 2180.37  4693.4 2178.72  4720.3 2176.63
  4733.8 2176.51  4763.2 2174.49    4769 2175.04  4778.9 2173.94  4800.3 2173.03
  4843.3 2172.47  4880.4 2169.76  4896.1 2169.81  4923.3 2168.59  4944.8 2169.04
  4962.7 2168.38  4966.3 2167.92    4989  2169.3  4997.4 2165.41  5005.8    2165
  5006.3  2164.5  5015.3  2164.5  5015.8    2165    5021 2168.77  5039.9 2171.73
  5051.8 2175.17  5062.1 2176.29  5123.7 2179.05  5130.5 2180.25  5154.5 2180.76
#Mann= 5 ,-1 , 0
  4536.6     .07       0  4693.4     .16       0  4962.7     .07       0
  5005.8     .07       0  5015.8     .07       0
Bank Sta=5005.8,5015.8
XS Rating Curve= 0 ,0
Exp/Cntr=0.3,0.1

Type RM Length L Ch R = 1 ,4030    ,496,496,496
BEGIN DESCRIPTION:
Idlewild Creek 6.0
END DESCRIPTION:
XS GIS Cut Line= 3
      1371255.03      6844038.03       1370889.2      6843736.94
      1370554.96      6843687.99
#Sta/Elev= 30
  4526.2 2186.68  4533.4 2186.14  4554.2  2181.9  4582.9 2179.84  4689.8 2177.23
  4710.6 2177.85  4774.5 2176.71  4891.6 2170.52  4938.7 2169.39  4959.6 2166.59
  4966.6 2167.04  4980.4 2165.43  4988.2 2162.68  4994.3 2162.15  4994.8 2161.65
  5004.7 2162.15  5017.2 2162.94  5023.3 2163.59  5028.4 2162.17  5044.7 2164.28
  5064.9 2164.23    5075 2162.87  5085.1 2166.98  5093.2  2172.3  5098.2 2171.44
  5125.5 2173.72  5226.6 2178.42  5256.9 2181.85  5302.8 2192.04  5337.8 2194.59
#Mann= 5 ,-1 , 0
  4526.2     .07       0  4891.6     .16       0  4994.3     .07       0
  5004.7     .16       0  5017.2     .07       0
Bank Sta=4994.3,5004.7
XS Rating Curve= 0 ,0
Exp/Cntr=0.3,0.1

Type RM Length L Ch R = 1 ,3534    ,419,419,419
BEGIN DESCRIPTION:
Idlewild Creek 5.0
END DESCRIPTION:
XS GIS Cut Line= 3
      1371155.01      6843638.02      1371006.46      6843291.52
        1371005.      6843188.03
#Sta/Elev= 30
    4623 2176.84  4666.5 2175.72  4690.1 2174.21  4699.2 2174.89  4713.7 2173.06
  4731.8 2172.84  4766.3 2170.08  4823.8 2167.46    4837 2167.76  4873.3 2166.67
  4884.1 2167.56  4889.5 2166.66  4905.9 2166.64  4942.1 2167.66  4960.2 2166.72
  4965.7 2165.87  4971.2 2164.09  4980.7  2162.9  4993.9 2161.17  4994.4 2160.67
    5004 2160.67  5004.5 2161.17  5013.5 2161.86  5023.5 2166.76  5043.5 2178.01
  5053.5 2185.84  5063.5 2192.34  5093.5 2195.75    5101 2197.53  5103.5 2197.53
#Mann= 5 ,-1 , 0
    4623     .07       0  4823.8     .16       0  4980.7     .07       0
  4993.9     .07       0  5004.5     .16       0
Bank Sta=4993.9,5004.5
XS Rating Curve= 0 ,0
Exp/Cntr=0.3,0.1

Type RM Length L Ch R = 1 ,3115    ,181,181,181
BEGIN DESCRIPTION:
Idlewild Creek 4.1
END DESCRIPTION:
XS GIS Cut Line= 3
      1371788.96      6843972.58       1371407.7      6843332.64
      1371125.26      6842852.68
#Sta/Elev= 30
  4255.1 2200.84  4255.6 2200.84  4283.7 2198.34  4327.8 2188.72  4364.8  2182.9
  4370.7 2183.76  4407.7  2179.1  4436.2  2178.7  4625.7 2172.03  4807.1 2169.72
  4934.7 2169.06  4960.5 2164.97  5004.9 2160.87  5013.6 2159.64  5014.1 2159.14
  5024.3 2159.64  5154.2 2163.64    5183 2164.47  5257.8 2167.88  5306.1 2174.01
  5341.9 2176.43  5399.9 2185.89  5423.1 2190.98  5429.1 2195.25  5434.9 2193.43
  5450.5 2196.41  5466.2 2202.83  5481.1  2205.1  5532.8  2206.9  5556.9 2206.04
#Mann= 12 ,-1 , 0
  4255.1     .07       0  4255.6    .035       0  4436.2     .07       0
  4807.1     .16       0  4934.7     .07       0  5004.9     .16       0
  5013.6     .07       0  5024.3     .16       0  5154.2     .07       0
    5183     .16       0  5257.8     .07       0  5532.8    .035       0
Bank Sta=5013.6,5024.3
XS Rating Curve= 0 ,0
Exp/Cntr=0.3,0.1

Type RM Length L Ch R = 1 ,2934    ,393,393,393
BEGIN DESCRIPTION:
Idlewild Creek 4.0
END DESCRIPTION:
XS GIS Cut Line= 3
      1371940.64       6843914.4      1371839.87      6843749.17
      1371286.11      6842825.13
#Sta/Elev= 30
  4148.8  2192.2  4165.7 2190.42  4171.6  2191.8  4190.8 2188.58  4238.3 2183.35
  4275.8 2181.58  4542.2 2169.82  4689.9 2167.57  4796.2 2168.84  4860.9 2164.62
    4980 2160.41  5002.9 2159.24  5067.1 2160.58  5119.6 2159.63  5120.1 2158.53
  5120.6 2158.03  5130.8 2158.53  5177.9 2160.88  5183.8 2162.88  5193.5 2163.31
  5199.3 2165.68  5214.9 2166.65  5236.3  2170.3    5279 2183.15  5294.6 2183.44
    5323 2189.54  5347.5 2189.16  5368.5  2186.8  5389.8 2187.51  5419.6 2192.39
#Mann= 9 ,-1 , 0
  4148.8     .07       0  4190.8    .035       0  4275.8     .07       0
  4796.2     .16       0  4860.9     .07       0    4980     .16       0
  5120.1     .07       0  5130.8     .16       0  5347.5     .07       0
Bank Sta=5120.1,5130.8
XS Rating Curve= 0 ,0
Exp/Cntr=0.3,0.1
