--- Long Branch.prj (project) ---

Proj Title=Long Branch Base Level Engineering
Current Plan=p01
Default Exp/Contr=0.3,0.1
English Units
Geom File=g01
Flow File=f01
Plan File=p01
Y Axis Title=Elevation
X Axis Title(PF)=Main Channel Distance
X Axis Title(XS)=Station
BEGIN DESCRIPTION:
Long Branch
END DESCRIPTION:
DSS Export Rating Curves= 0
DSS Export Rating Curve Sorted= 0
DSS Export Volume Flow Curves= 0
DXF OffsetX= 0
DXF OffsetY= 0
DXF ScaleX= 1
DXF ScaleY= 10

--- Long Branch.p01 (plan) ---

Plan Title=Multiple Run
Short Identifier=Multiple
Geom File=g01
Flow File=f01
Subcritical Flow
K Sum by GR= 0
Std Step Tol= 0.01
Critical Tol= 0.01
Num of Std Step Trials= 20
Max Error Tol= 0.3
Flow Tol Ratio= 0.001
Split Flow NTrial= 30
Split Flow Tol= 0.02
Split Flow Ratio= 0.02
Log Output Level= 0
Friction Slope Method= 1
Unsteady Friction Slope Method= 2
Unsteady Bridges Friction Slope Method= 1
Parabolic Critical Depth
Global Vel Dist=  1 , 1 , 1
Global Log Level= 0
CheckData=True
Encroach Param= -1, 0, 0, 0
BEGIN DESCRIPTION:
Multiple Run
END DESCRIPTION:

--- Long Branch.f01 (steady flow) ---

Flow Title=Multiple
Number of Profiles=7
Profile Names=10-year,25-year,50-year,1pct_min,100-year,1pct_plu,500-year
River Rch & RM= Long Branch,Reach-1,49613
     135     180     215     128     255     508     362
River Rch & RM= Long Branch,Reach-1,48620
     197     267     321     192     383     765     553
River Rch & RM= Long Branch,Reach-1,38838
     244     332     401     240     480     957     696
River Rch & RM= Long Branch,Reach-1,31944
     375     531     660     407     811    1619    1244
River Rch & RM= Long Branch,Reach-1,27224
     419     598     747     463     924    1844    1433
River Rch & RM= Long Branch,Reach-1,25267
     616     900    1145     720    1437    2868    2302
River Rch & RM= Long Branch,Reach-1,23815
     724    1069    1368     868    1731    3454    2813
River Rch & RM= Long Branch,Reach-1,21866
     767    1138    1461     929    1854    3700    3031
River Rch & RM= Long Branch,Reach-1,19878
     792    1178    1515     965    1926    3843    3159
River Rch & RM= Long Branch,Reach-1,18476
     829    1236    1592    1016    2028    4046    3337
River Rch & RM= Long Branch,Reach-1,17422
     844    1259    1623    1036    2067    4124    3404
River Rch & RM= Long Branch,Reach-1,15504
     891    1333    1723    1103    2200    4390    3641
River Rch & RM= Long Branch,Reach-1,10595
     903    1353    1750    1121    2236    4461    3704
River Rch & RM= Long Branch,Reach-1,8128
    1014    1517    1961    1255    2504    4996    4139
River Rch & RM= Long Branch,Reach-1,178
    1373    2080    2711    1748    3487    6957    5852
Boundary for River Rch & Prof#=Long Branch,Reach-1,1
Up Type=0
Dn Type=3
Dn Slope=0.005
Boundary for River Rch & Prof#=Long Branch,Reach-1,2
Up Type=0
Dn Type=3
Dn Slope=0.005
Boundary for River Rch & Prof#=Long Branch,Reach-1,3
Up Type=0
Dn Type=3
Dn Slope=0.005
Boundary for River Rch & Prof#=Long Branch,Reach-1,4
Up Type=0
Dn Type=3
Dn Slope=0.005
Boundary for River Rch & Prof#=Long Branch,Reach-1,5
Up Type=0
Dn Type=3
Dn Slope=0.005
Boundary for River Rch & Prof#=Long Branch,Reach-1,6
Up Type=0
Dn Type=3
Dn Slope=0.005
Boundary for River Rch & Prof#=Long Branch,Reach-1,7
Up Type=0
Dn Type=3
Dn Slope=0.005

--- Long Branch.g01 (geometry) ---

Geom Title=Existing Conditions
Program Version=4.10

River Reach=Long Branch     ,Reach-1
Reach XY= 30
        1348055.        6833738.      1346316.24      6834877.95
      1346363.04      6836591.32      1347518.33      6838601.33
      1349051.34      6839746.17      1349560.47      6841740.99
      1350594.05        6842328.      1351960.86      6845035.94
       1354958.3      6844929.92      1356160.45      6844190.18
      1357653.35       6844034.9      1358264.62      6843338.63
      1359199.22      6843735.92      1359851.57      6842445.79
      1361334.71      6843038.39       1361852.7      6842293.83
      1362854.01      6842484.47      1363510.85      6841739.49
      1365199.29      6842186.11        1365900.        6841933.
      1366102.53      6841093.45      1367278.99       6841015.7
      1367404.99      6840095.53      1368284.51      6840438.87
      1369043.41      6840139.38      1369384.64      6840688.39
      1370793.13      6839839.51      1371772.13      6840254.45
      1372302.45      6841182.27        1373955.        6841738.

Type RM Length L Ch R = 1 ,49613   ,993,993,993
BEGIN DESCRIPTION:
Long Branch 88.0
END DESCRIPTION:
XS GIS Cut Line= 3
      1346404.99      6833287.99      1347734.81        6833868.
      1349105.04      6834338.01
#Sta/Elev= 30
  3549.2 2414.29  3647.4 2413.97  3691.6 2414.65  3723.8 2413.74  3756.4 2413.59
  3936.7 2413.86    4117 2412.82  4163.8  2413.3  4192.9 2412.38  4536.3 2412.24
  4837.6 2411.99  5076.3  2411.8  5076.5  2411.3    5080  2411.3  5080.3  2411.8
  5416.9 2411.99  5505.5 2413.25  5581.7 2412.91  5661.8 2413.94  5761.4 2413.46
  5911.9 2414.44  6025.9 2414.13  6110.3 2414.86  6120.2 2415.51  6181.6 2415.27
  6205.4 2415.77  6226.6 2415.44  6258.3 2416.53  6300.6 2415.81  6448.6 2416.33
#Mann= 7 ,-1 , 0
  3549.2    .045       0  4536.3     .07       0  4837.6    .045       0
  5076.3    .045       0  5080.3    .045       0  6025.9    .035       0
  6181.6    .045       0
Bank Sta=5076.3,5080.3
XS Rating Curve= 0 ,0
Exp/Cntr=0.3,0.1

Type RM Length L Ch R = 1 ,48620   ,553,553,553
BEGIN DESCRIPTION:
Long Branch 87.0
END DESCRIPTION:
XS GIS Cut Line= 3
        1345405.        6832488.      1347405.57      6834488.25
      1349204.97        6834488.
#Sta/Elev= 30
    2171 2417.18  2199.3  2416.4  2401.6 2415.86  2418.9 2415.78  2531.6 2416.12
  2588.2 2414.92  2849.8 2414.51  3684.2 2413.92  3705.4 2414.52  3754.9 2413.77
  4009.5 2414.12  4087.3 2413.18  4320.6 2412.86  4940.9 2412.84  4941.1 2412.34
  4944.9 2412.84  5099.4 2413.85  5309.4 2413.33  5469.4 2414.63  5529.4 2413.97
  5739.4 2415.36  5789.4 2414.83  5989.4  2416.1  6049.4  2415.5    6240  2416.4
  6289.4  2417.1  6319.4 2415.87  6329.4  2416.8  6400.5 2416.39  6799.4 2416.85
#Mann= 7 ,-1 , 0
    2171    .045       0  2401.6     .07       0  2418.9    .045       0
  4940.9    .045       0  4944.9    .045       0    6240    .035       0
  6400.5    .045       0
Bank Sta=4940.9,4944.9
XS Rating Curve= 0 ,0
Exp/Cntr=0.3,0.1

Type RM Length L Ch R = 1 ,48067   ,1163,1163,1163
BEGIN DESCRIPTION:
Long Branch 4284
END DESCRIPTION:
XS GIS Cut Line= 3
      1345880.33      6833949.81      1346981.73      6834761.36
      1347895.99      6834626.89
#Sta/Elev= 30
  3631.9 2413.96  3662.5 2414.24  3948.2 2414.04  4020.8 2414.15  4041.6 2414.55
  4075.6 2413.97  4141.9    2414  4148.1 2413.71  4256.8 2414.01  4442.7 2413.66
  4507.2  2414.1  4549.1 2413.52  4563.8 2413.76    4570 2413.35  4929.3 2413.21
  4939.9 2412.84  4940.2 2412.34  4943.8 2412.34    4944 2412.84  4964.8 2413.17
  5185.2 2413.21  5225.7 2413.73  5541.3 2413.42  5549.1 2413.86  5579.4 2413.88
    5606 2413.53  5680.8 2413.99  5710.8 2414.71  5740.4    2414  5924.1 2414.49
#Mann= 3 ,-1 , 0
  3631.9    .045       0  4939.9    .045       0    4944    .045       0
Bank Sta=4939.9,4944
XS Rating Curve= 0 ,0
Exp/Cntr=0.3,0.1

Type RM Length L Ch R = 1 ,46904   ,676,676,676
BEGIN DESCRIPTION:
Long Branch 4283
END DESCRIPTION:
XS GIS Cut Line= 3
       1345479.3      6834158.15       1346216.4      6835178.08
      1347734.48      6834725.86
#Sta/Elev= 30
  3741.6 2413.55  4082.5 2413.94  4360.9 2413.37  4396.5 2412.95  4469.4 2413.42
  4511.8 2412.65  4863.8 2412.36  5113.3 2412.64  5132.1  2412.3  5132.4  2411.8
    5136  2411.8  5136.3  2412.3  5290.7 2412.68    5322 2412.35    5395 2412.56
  5434.8 2413.12  5551.6 2412.67  5708.1 2413.21  5916.8 2413.21  5958.4 2413.86
  6035.2 2413.27    6115 2413.74    6173 2413.75    6188 2413.37  6396.7 2413.83
  6415.6 2414.42  6420.9 2414.02  6438.5 2414.71  6487.2 2414.04    6584 2414.24
#Mann= 3 ,-1 , 0
  3741.6    .045       0  5132.1    .045       0  5136.3    .045       0
Bank Sta=5132.1,5136.3
XS Rating Curve= 0 ,0
Exp/Cntr=0.3,0.1

Type RM Length L Ch R = 1 ,46228   ,989,989,989
BEGIN DESCRIPTION:
Long Branch 86.0
END DESCRIPTION:
XS GIS Cut Line= 3
      1345005.01      6833938.01      1346221.59      6835721.48
      1348004.99      6834738.01
#Sta/Elev= 30
  2841.1  2413.5  3031.8 2413.43  3247.5 2413.56  3740.1  2413.7  4000.3  2413.1
  4027.4 2413.58    4087 2412.77  4784.1 2412.34  4813.9 2412.85  4834.9 2412.17
  4891.8 2411.74  4991.4 2411.55  4991.7 2411.05  4995.3 2411.05  4995.6 2411.55
  5100.7 2411.85  5152.4 2412.81    5198 2412.26  5460.7 2412.52    5519 2413.19
  5572.9 2412.76  5779.3  2412.8  6020.3 2413.61  6382.1 2413.93  6447.5 2414.72
  6499.9 2414.19  6682.6  2414.5  6800.5 2415.51  6838.3 2414.84  7036.6  2415.2
#Mann= 5 ,-1 , 0
  2841.1    .045       0  3031.8     .07       0  3247.5    .045       0
  4991.4    .045       0  4995.6    .045       0
Bank Sta=4991.4,4995.6
XS Rating Curve= 0 ,0
Exp/Cntr=0.3,0.1

Type RM Length L Ch R = 1 ,45239   ,469,469,469
BEGIN DESCRIPTION:
Long Branch 85.0
END DESCRIPTION:
XS GIS Cut Line= 3
      1344604.96      6835837.99      1346405.41       6836460.7
        1348205.        6834638.
#Sta/Elev= 30
  3094.9 2412.15  3198.7 2412.15    3204 2411.54  3229.9 2411.83  3235.2 2411.11
  3266.4 2410.88    3474 2410.35  4211.4 2410.07  4304.9 2410.82    4407  2409.5
    4995 2408.48  4995.3 2407.98  4999.2 2408.48  5249.1 2409.33  5305.7 2410.38
  5482.4 2410.55  5517.8 2411.38  5602.7 2411.09  5878.4 2411.74  5963.3 2412.79
  6083.5  2412.4  6514.9 2413.71  6571.4 2413.97  6599.7 2414.93    6628 2414.16
  6847.2 2414.66  6875.5 2415.53  6939.2 2414.89  7448.3 2415.08  7561.4 2415.99
#Mann= 3 ,-1 , 0
  3094.9    .045       0    4995    .045       0  4999.2    .045       0
Bank Sta=4995,4999.2
XS Rating Curve= 0 ,0
Exp/Cntr=0.3,0.1

Type RM Length L Ch R = 1 ,44770   ,498,498,498
BEGIN DESCRIPTION:
Long Branch 84.0
END DESCRIPTION:
XS GIS Cut Line= 3
      1344554.97      6836037.99      1346552.85      6836843.89
        1348155.        6834838.
#Sta/Elev= 30
  2845.7 2409.97  4012.1 2409.99  4138.3 2409.53  4143.6 2407.89  4167.8 2409.42
  4191.9 2408.06  4197.3 2409.68  4221.5 2408.74  4290.6 2409.22  4299.3 2409.08
  4304.7 2407.15  4328.9 2409.09  4344.6  2407.4  4358.4 2408.96  4382.5 2409.24
  4804.8 2407.76  5062.3 2407.51    5120  2409.1  5132.3 2406.35  5132.5 2405.85
  5136.5 2406.35  5148.3 2408.42  5161.6 2407.57  5446.6 2408.33  5731.6 2410.44
  6500.1 2412.96  6543.3 2414.03    6657 2413.57  6748.2 2414.86  7567.2 2416.23
#Mann= 5 ,-1 , 0
  2845.7    .045       0  4804.8    .035       0  5062.3    .045       0
  5132.3    .035       0  5136.5    .045       0
Bank Sta=5132.3,5136.5
XS Rating Curve= 0 ,0
Exp/Cntr=0.3,0.1

Type RM Length L Ch R = 1 ,44272   ,498,498,498
BEGIN DESCRIPTION:
Long Branch 83.0
END DESCRIPTION:
XS GIS Cut Line= 3
       1345097.8      6836936.58      1346756.65      6837234.02
      1347954.99      6835438.01
#Sta/Elev= 30
  3314.7 2407.63  3579.4 2408.29  3697.9 2407.25  4500.5 2406.99  4543.6  2407.7
  4663.1  2406.4  4866.3 2406.87  5022.5 2405.11  5022.8 2404.61  5026.8 2405.11
  5337.3 2406.51    5352 2406.25  5457.3 2406.62  5478.3 2407.79  5493.3 2405.24
  5500.1 2407.77  5508.3 2407.91  5536.2 2406.89  5868.8 2407.89  5904.9 2409.02
  6034.1 2408.91  6136.2 2410.35  6271.4 2410.32  6316.4 2411.46  6343.5 2410.82
  6532.7 2411.88  6553.8 2412.78  6755.1 2413.04  6776.1 2414.09  7159.1 2414.99
#Mann= 5 ,-1 , 0
  3314.7    .045       0  5022.5    .045       0  5026.8    .045       0
  5337.3    .035       0    5352    .045       0
Bank Sta=5022.5,5026.8
XS Rating Curve= 0 ,0
Exp/Cntr=0.3,0.1

Type RM Length L Ch R = 1 ,43774   ,498,498,498
BEGIN DESCRIPTION:
Long Branch 82.0
END DESCRIPTION:
XS GIS Cut Line= 3
      1345429.86      6838163.97      1347131.78      6837514.32
        1347955.        6835738.
#Sta/Elev= 30
  3178.3 2406.17  3493.4 2406.16  3600.6 2406.31  3628.8 2406.43  3651.4 2402.78
  3651.7 2402.28  3655.7 2402.78  3665.5 2405.56  3683.6  2406.6  3927.1 2405.39
  4049.1 2405.18  4106.9 2405.85  4211.4 2404.18  4421.1 2403.83  5361.3 2403.74
  5512.3 2404.17  5581.5 2405.45  5633.8 2405.45  5656.7 2406.87  5668.3 2404.86
  5679.3    2407  5690.6 2407.11  5701.3 2405.66  5828.1 2406.35  6251.6 2409.12
  6428.8 2411.47  6588.9 2411.76  6627.2 2412.88  6649.2 2412.16  6957.8  2414.2
#Mann= 12 ,-1 , 0
  3178.3    .035       0  3493.4    .045       0  3600.6     .07       0
  3651.4     .07       0  3655.7     .07       0  3927.1    .045       0
  4049.1     .07       0  4106.9    .045       0  4421.1     .07       0
  5361.3    .045       0  5512.3    .035       0  5581.5    .045       0
Bank Sta=3651.4,3655.7
XS Rating Curve= 0 ,0
Exp/Cntr=0.3,0.1

Type RM Length L Ch R = 1 ,43276   ,1036,1036,1036
BEGIN DESCRIPTION:
Long Branch 81.0
END DESCRIPTION:
XS GIS Cut Line= 3
        1345405.        6839288.      1347225.16      6837888.32
      1348159.64      6835973.03
#Sta/Elev= 30
  2703.9 2410.05  2839.8 2410.54    3224 2408.88  3296.6 2409.98  3373.5 2408.24
  3464.7 2408.62  3510.4 2406.94  3605.6 2406.62    3937 2403.76  4465.5 2404.02
    4480  2403.2  4483.6 2401.77    4484 2401.27    4489 2401.77  4507.8 2404.21
  4864.2 2403.15  5709.6 2404.14  5817.1 2403.91  5970.5  2404.4  6010.9 2406.34
    6024 2404.87  6033.4 2406.72  6046.3 2406.83    6056 2404.77  6068.5 2406.18
  6517.7 2409.08  6697.9 2411.67  7018.9 2412.83  7047.7 2414.08  7131.1 2413.59
#Mann= 9 ,-1 , 0
  2703.9    .045       0  3464.7     .07       0  3605.6    .035       0
    3937     .07       0  4483.6     .07       0    4489     .07       0
  5709.6    .045       0  5817.1    .035       0  5970.5    .045       0
Bank Sta=4483.6,4489
XS Rating Curve= 0 ,0
Exp/Cntr=0.3,0.1

Type RM Length L Ch R = 1 ,42240   ,148,148,148
BEGIN DESCRIPTION:
Long Branch 80.0
END DESCRIPTION:
XS GIS Cut Line= 3
      1347223.39      6839581.02      1347521.39      6838604.79
      1347999.89      6836457.04
#Sta/Elev= 30
  3979.3 2410.09    4780 2406.31    5358 2405.89  5581.6  2405.1  5734.4 2405.99
  5744.6 2405.49  5762.4    2402  5762.8  2401.5  5767.8    2402  5772.8 2404.88
  5777.9 2402.63  5785.6 2405.75  5864.9 2404.03  6112.3 2404.47  6267.1 2404.51
  6281.8 2405.47  6417.4 2404.64    6466 2405.64  6509.5 2404.82  6514.6 2405.92
    6553 2405.07  6601.6 2407.56  6615.4 2404.48  6625.7 2404.97  6635.9 2407.63
  6650.2 2407.72  6666.7 2405.86  6676.9 2407.36  6755.1 2407.42  7200.4 2410.25
#Mann= 8 ,-1 , 0
  3979.3    .045       0    4780     .07       0    5358    .094       0
  5581.6     .07       0  5762.4     .07       0  5767.8     .07       0
  6112.3    .035       0  6755.1    .045       0
Bank Sta=5762.4,5767.8
XS Rating Curve= 0 ,0
Exp/Cntr=0.3,0.1

Type RM Length L Ch R = 1 ,42092   ,303,303,303
BEGIN DESCRIPTION:
Long Branch 79.0
END DESCRIPTION:
XS GIS Cut Line= 3
      1347423.57      6839542.41      1347636.54      6838688.67
      1348389.07      6836521.72
#Sta/Elev= 30
  4120.1 2409.32  4396.2 2407.48  4454.5 2407.75    4520 2406.69  4578.1 2407.53
    4609 2406.12  5163.5 2405.97  5375.4  2406.2  5492.6 2406.55  5739.3 2406.52
  5786.1 2407.18  5837.9 2407.68  5847.6 2405.86  5855.5 2401.76  5855.9 2401.26
  5860.9 2401.76  5869.1 2403.08  5879.3 2407.14  5911.1 2406.18  5953.6 2406.79
  6334.5 2406.72  6444.5 2408.36  6594.8 2408.56    6657 2410.01  6719.2  2409.3
  6863.8 2409.88  6874.8 2410.93  6954.7  2411.6    7232 2412.57  7293.9 2412.78
#Mann= 10 ,-1 , 0
  4120.1    .035       0  5163.5    .094       0  5375.4    .035       0
  5492.6    .045       0  5786.1    .035       0  5855.5    .035       0
  5860.9    .035       0  5953.6    .045       0  6954.7    .035       0
    7232    .045       0
Bank Sta=5855.5,5860.9
XS Rating Curve= 0 ,0
Exp/Cntr=0.3,0.1

Type RM Length L Ch R = 1 ,41789   ,499,499,499
BEGIN DESCRIPTION:
Long Branch 78.0
END DESCRIPTION:
XS GIS Cut Line= 3
      1347407.77      6839642.77       1347907.3      6838793.83
      1348261.78      6837991.33
#Sta/Elev= 30
    4015 2409.67  4171.4 2408.56  4198.6 2409.11  4206.6 2408.88  4345.4 2407.41
  4368.6 2407.28    4390 2407.76  4438.8  2406.5  4454.4 2406.43  4491.5 2407.47
    4513 2406.29  4534.5 2405.94  4555.9 2406.48  4645.8 2405.64  4920.3 2405.45
  4920.8 2404.95  4925.4 2404.95  4925.8 2405.45  4950.4 2405.81  4987.5  2405.5
  5154.6 2405.87  5192.2 2406.49  5380.7  2406.4  5432.8 2407.18    5474 2406.85
  5572.6 2407.42  5662.3 2407.23  5684.2 2407.62  5809.4 2407.97  5877.3 2408.58
#Mann= 5 ,-1 , 0
    4015    .035       0  4206.6    .045       0  4920.3    .045       0
  4925.8    .045       0  5809.4    .035       0
Bank Sta=4920.3,4925.8
XS Rating Curve= 0 ,0
Exp/Cntr=0.3,0.1

Type RM Length L Ch R = 1 ,41290   ,475,475,475
BEGIN DESCRIPTION:
Long Branch 77.0
END DESCRIPTION:
XS GIS Cut Line= 3
      1347467.67      6839671.41       1348298.5      6839081.25
      1348532.72      6838047.97
#Sta/Elev= 30
  3980.9 2409.14    4039 2408.89  4075.7 2409.39  4132.3 2408.39  4268.8 2408.18
  4274.9 2407.74  4319.2 2407.63  4346.3 2406.83  4375.8 2407.83  4390.6 2406.69
  4411.5 2406.05  4476.7 2406.37  4541.9 2405.45  4862.9 2405.12  4919.2 2404.66
  4919.6 2404.16  4924.3 2404.16  4924.7 2404.66  5310.9 2405.86  5341.7 2406.53
  5373.1 2406.19  5550.8 2406.65  5577.5 2407.42  5618.6 2406.99  5782.6  2407.4
  5819.8 2408.17  5844.1 2407.74  6008.2 2408.15  6045.5 2408.75  6059.5 2408.65
#Mann= 4 ,-1 , 0
  3980.9    .045       0  4919.2    .045       0  4924.7    .045       0
  6045.5    .035       0
Bank Sta=4919.2,4924.7
XS Rating Curve= 0 ,0
Exp/Cntr=0.3,0.1

Type RM Length L Ch R = 1 ,40815   ,493,493,493
BEGIN DESCRIPTION:
Long Branch 76.0
END DESCRIPTION:
XS GIS Cut Line= 3
      1346755.03      6839887.99      1348534.97      6839468.07
      1348705.88       6838085.4
#Sta/Elev= 30
  3171.2 2410.89  3688.6 2409.98  3746.5 2410.75  3760.5 2409.01  3767.1 2410.19
    3791  2410.4  3802.9 2411.47  3808.2  2409.9  3887.6 2409.32  3993.1 2409.51
  4019.6 2408.69  4241.5 2407.39  4270.5 2407.92  4445.2  2404.6  4453.1 2405.05
  4458.3  2404.4    4476 2405.13  4542.9 2403.48  4558.2 2404.44  4619.9 2403.56
  4650.7 2404.51  4702.1 2403.35  4994.6 2401.68  4995.1 2401.18  5000.2 2401.68
  5367.5 2404.96  5644.9 2405.36  5691.7 2406.25  6346.7  2408.4  6393.2 2408.63
#Mann= 7 ,-1 , 0
  3171.2    .045       0  3688.6    .094       0    3791    .035       0
  3887.6    .045       0  4994.6    .045       0  5000.2    .045       0
  6346.7    .035       0
Bank Sta=4994.6,5000.2
XS Rating Curve= 0 ,0
Exp/Cntr=0.3,0.1

Type RM Length L Ch R = 1 ,40322   ,496,496,496
BEGIN DESCRIPTION:
Long Branch 75.0
END DESCRIPTION:
XS GIS Cut Line= 3
      1347155.04      6840487.98      1348953.31      6839692.15
      1349122.86       6838175.5
#Sta/Elev= 30
  3033.5  2411.9  3047.8  2410.8  3055.3 2412.06  3088.1 2410.85  3099.9 2411.98
  3123.2 2410.78    3260 2410.36  3580.2 2409.52  3738.2 2407.97    3767 2408.46
  3798.9 2407.36  3906.7 2406.88  3982.1 2405.34  4086.2 2405.17  4156.1 2403.77
    4291 2403.38  4323.9 2402.31  4509.8  2401.6  4542.6 2400.65    4919 2399.75
  4919.5 2399.25  4924.7 2399.75  5155.2 2400.24    5467 2403.52  5929.9 2405.26
  6000.3 2406.27  6171.4 2406.67  6221.7 2407.74  6487.2 2408.21  6526.1  2408.7
#Mann= 5 ,-1 , 0
  3033.5    .035       0    3260    .045       0    4919    .045       0
  4924.7    .045       0  6487.2    .035       0
Bank Sta=4919,4924.7
XS Rating Curve= 0 ,0
Exp/Cntr=0.3,0.1

Type RM Length L Ch R = 1 ,39826   ,988,988,988
BEGIN DESCRIPTION:
Long Branch 74.0
END DESCRIPTION:
XS GIS Cut Line= 3
        1347355.        6841488.      1349138.19      6840071.39
      1350098.88      6838386.42
#Sta/Elev= 30
  2722.6 2414.72  2790.5 2413.43  2850.3 2412.91  2872.4 2413.82  2907.6 2412.39
  2923.8  2412.6  3049.3 2411.82  3178.7 2410.96  3463.4 2409.09  3519.6 2407.81
  3577.3 2407.99  3633.3 2406.26    3683 2406.52  3718.8 2405.04  3782.6 2404.87
  3819.2 2403.51  3875.2 2402.96  3904.1 2403.23  3932.9 2402.03  4025.3 2401.74
  4061.1 2400.53  4245.3 2400.26  4331.8 2399.09  4790.3 2398.63  4790.8 2398.13
    4796 2398.63  5270.3 2399.16  5748.5 2402.58  6917.5 2407.63  6939.6 2407.87
#Mann= 8 ,-1 , 0
  2722.6    .035       0  2790.5     .07       0  2923.8    .045       0
  3049.3     .07       0  3178.7    .045       0  4790.3    .045       0
    4796    .045       0  6917.5    .035       0
Bank Sta=4790.3,4796
XS Rating Curve= 0 ,0
Exp/Cntr=0.3,0.1

Type RM Length L Ch R = 1 ,38838   ,499,499,499
BEGIN DESCRIPTION:
Long Branch 73.0
END DESCRIPTION:
XS GIS Cut Line= 3
      1347755.03      6841837.98      1349357.84      6840893.87
      1350355.02      6838887.96
#Sta/Elev= 30
  3139.8 2413.41  3233.4 2412.62  3270.5 2413.58    3292 2412.27  3418.3 2411.08
  3453.1  2412.1  3489.2 2410.33  3569.2 2410.73  3592.4 2409.17  3659.1 2408.24
  3696.2  2408.9  3776.2 2406.88  3803.5 2407.57  3840.6 2405.85  3899.1 2404.94
    3929 2405.65  3973.4 2403.69  4161.1 2401.81  4229.1 2400.01  4277.8 2400.39
  4309.1 2399.37  4484.8 2398.62  4912.3 2398.24  4912.8 2397.74  4918.6 2398.24
  5994.1 2399.01  6480.7 2401.82  6525.3 2402.77  7186.8 2405.16  7240.1 2406.08
#Mann= 3 ,-1 , 0
  3139.8    .045       0  4912.3    .045       0  4918.6    .045       0
Bank Sta=4912.3,4918.6
XS Rating Curve= 0 ,0
Exp/Cntr=0.3,0.1

Type RM Length L Ch R = 1 ,38339   ,499,499,499
BEGIN DESCRIPTION:
Long Branch 72.0
END DESCRIPTION:
XS GIS Cut Line= 3
        1347905.        6842088.      1349491.35      6841274.67
      1351305.02      6839487.98
#Sta/Elev= 30
  3217.3  2414.3  3374.6 2412.61  3403.2 2413.89    3431  2412.3  3520.7 2411.39
  3558.5 2412.27  3597.3 2410.24  3663.9 2410.73  3736.1 2408.29  3767.9 2409.14
  3802.7 2407.22  3880.3 2407.46    3914 2405.75  4003.9  2405.5  4041.3 2403.91
  4138.8  2403.6  4174.4 2401.93  4374.8 2399.63  4975.7  2397.9  4976.2  2397.4
  4982.1  2397.9  5331.6 2398.55  5480.1 2398.46    5573 2398.48  5615.8  2398.4
  5716.1 2398.67  5751.5 2398.64  6172.7 2400.22  6507.1 2401.57  7545.9 2405.47
#Mann= 11 ,-1 , 0
  3217.3    .045       0  4975.7    .045       0  4982.1    .045       0
  5331.6     .07       0  5480.1    .035       0    5573     .07       0
  5615.8    .035       0  5716.1     .07       0  5751.5    .035       0
  6172.7     .07       0  6507.1    .045       0
Bank Sta=4975.7,4982.1
XS Rating Curve= 0 ,0
Exp/Cntr=0.3,0.1

Type RM Length L Ch R = 1 ,37840   ,492,492,492
BEGIN DESCRIPTION:
Long Branch 71.0
END DESCRIPTION:
XS GIS Cut Line= 3
        1348105.        6842038.      1349554.57      6841706.49
      1351155.01      6839687.99
#Sta/Elev= 30
    3513 2413.87    3554 2412.13  3646.4 2411.23    3671 2412.25  3713.9 2410.15
    3790  2410.5    3831 2408.75  4029.9 2407.41  4138.8 2404.71  4163.9 2405.71
  4261.9 2402.92    4303 2403.59  4345.9 2401.77  4415.7 2402.12  4456.8 2400.47
  4549.1 2400.48  4579.9 2399.06  5103.6 2397.64  5387.9 2397.49  5388.4 2396.99
  5394.4 2397.49  5902.3 2398.45  5969.6 2398.51  6162.8 2398.74  6214.1 2399.36
  6336.4 2399.88  6511.6    2401  6797.4 2402.09    7064 2402.05    7576 2404.75
#Mann= 11 ,-1 , 0
    3513    .045       0  5103.6     .07       0  5387.9    .045       0
  5394.4     .07       0  5902.3    .035       0  5969.6     .07       0
  6162.8    .035       0  6214.1     .07       0  6336.4    .035       0
  6511.6     .07       0  6797.4    .045       0
Bank Sta=5387.9,5394.4
XS Rating Curve= 0 ,0
Exp/Cntr=0.3,0.1

Type RM Length L Ch R = 1 ,37348   ,496,496,496
BEGIN DESCRIPTION:
Long Branch 70.0
END DESCRIPTION:
XS GIS Cut Line= 3
      1348254.97      6842338.01      1349836.75      6841988.19
      1351255.03      6840187.96
#Sta/Elev= 30
    3380 2412.98  3431.2 2413.68  3564.4 2411.08  3589.2 2412.22  3625.8 2410.46
    3718 2409.64  3738.5 2410.72    3774 2408.92  4002.4 2407.41  4117.4  2404.7
  4143.6 2405.63  4187.2  2403.8  4284.7 2403.56  4333.5  2401.7  4486.1 2399.94
  5059.5 2397.78  5080.9 2397.59  5081.4 2397.09  5088.1 2397.59  5711.5 2397.74
  6257.7 2400.07  6434.2 2401.37  6535.6  2401.1  6680.8 2401.34  6711.8 2401.39
  6796.4 2402.02  6877.9 2401.78  6980.9 2401.85  7162.4 2402.98  7291.8 2403.43
#Mann= 13 ,-1 , 0
    3380    .045       0  5059.5     .07       0  5080.9    .045       0
  5088.1     .07       0  6257.7    .035       0  6434.2     .07       0
  6535.6    .035       0  6680.8     .07       0  6711.8    .035       0
  6796.4     .07       0  6877.9    .035       0  6980.9     .07       0
  7162.4    .045       0
Bank Sta=5080.9,5088.1
XS Rating Curve= 0 ,0
Exp/Cntr=0.3,0.1

Type RM Length L Ch R = 1 ,36852   ,1492,1492,1492
BEGIN DESCRIPTION:
Long Branch 69.0
END DESCRIPTION:
XS GIS Cut Line= 3
      1348404.99      6843138.01      1350188.57      6842120.31
      1351405.03      6840337.96
#Sta/Elev= 30
  2946.5 2412.64  3143.1 2410.99  3165.3 2412.02  3349.5 2409.55  3379.3  2410.5
    3407 2409.01  3556.5 2408.98  3707.7 2406.61  3745.1 2407.44  3782.6 2405.91
    3928 2405.35  3965.5 2403.85  4089.3 2403.57  4126.8 2401.83  4207.4  2402.2
  4244.9 2400.61  4368.7 2400.53  4406.2 2399.16  4631.8  2398.9  4854.8 2397.98
  4855.3 2397.48    4862 2397.98  5747.5 2398.62  6086.7 2400.21  6156.2 2400.41
  6255.9 2400.55  6742.4 2401.57    6965 2402.33  7091.4 2402.99  7157.9 2403.73
#Mann= 10 ,-1 , 0
  2946.5    .045       0  4631.8     .07       0  4854.8     .07       0
    4862     .07       0  6086.7    .035       0  6156.2     .07       0
  6255.9    .035       0  6742.4     .07       0    6965    .035       0
  7091.4    .045       0
Bank Sta=4854.8,4862
XS Rating Curve= 0 ,0
Exp/Cntr=0.3,0.1

Type RM Length L Ch R = 1 ,35360   ,495,495,495
BEGIN DESCRIPTION:
Long Branch 68.0
END DESCRIPTION:
XS GIS Cut Line= 3
      1348755.01        6843088.      1350735.27      6842867.49
        1350955.        6841088.
#Sta/Elev= 30
  3007.5 2409.93  3037.7 2409.48  3057.8 2410.39    3088  2409.1  3188.6 2407.97
  3218.8    2409    3249 2407.44  3369.7 2406.62  3409.5 2407.26  3450.2 2405.94
  3570.9 2404.74  3601.1 2405.64  3631.3 2404.25    3742 2402.89  3762.1 2403.85
  3802.4 2402.05    3903 2401.87  3933.2 2400.61  4069.9 2399.75  4305.5 2398.34
  4404.5 2398.85  4446.3 2397.91  4707.9 2398.13  4965.9 2396.89  4966.4 2396.39
  4973.2 2396.89  6420.9 2399.85  6545.4 2400.22  6780.1 2400.88    6793 2401.32
#Mann= 7 ,-1 , 0
  3007.5    .045       0  4069.9     .07       0  4965.9     .07       0
  4973.2     .07       0  6420.9    .035       0  6545.4     .07       0
  6780.1    .035       0
Bank Sta=4965.9,4973.2
XS Rating Curve= 0 ,0
Exp/Cntr=0.3,0.1

Type RM Length L Ch R = 1 ,34865   ,496,496,496
BEGIN DESCRIPTION:
Long Branch 67.0
END DESCRIPTION:
XS GIS Cut Line= 3
      1349154.97        6843088.      1350955.41      6843283.28
        1351755.        6841488.
#Sta/Elev= 30
    3189 2407.46  3229.3 2405.98    3360 2404.73  3390.2 2405.54  3509.7 2403.27
  3561.2 2403.93  3591.4 2402.37  3932.3 2399.26  4305.5 2397.82  4355.8  2396.7
  4738.1  2396.4  4965.7 2393.24  4966.2 2392.74  4973.1 2393.24  5057.7 2394.14
  5093.4 2395.83  5231.3  2395.7  5268.5 2397.22  5290.4 2396.33  5526.6 2397.87
  5739.2 2397.35    5783 2398.61  5821.9  2397.6    5990 2397.96  6024.2 2399.11
  6238.8 2398.71  6275.6 2399.87  6725.4 2399.58  6755.2 2399.56  6965.3 2399.86
#Mann= 6 ,-1 , 0
    3189    .045       0  3932.3     .07       0  4965.7     .07       0
  4973.1     .07       0  6725.4    .035       0  6755.2     .07       0
Bank Sta=4965.7,4973.1
XS Rating Curve= 0 ,0
Exp/Cntr=0.3,0.1

Type RM Length L Ch R = 1 ,34369   ,496,496,496
BEGIN DESCRIPTION:
Long Branch 66.0
END DESCRIPTION:
XS GIS Cut Line= 3
      1349054.97        6843538.      1351054.55      6843747.28
      1352055.02      6841937.96
#Sta/Elev= 30
  2989.5  2408.1  3059.9 2407.61  3129.4 2405.47  3134.5 2406.64  3170.5 2405.02
  3210.7 2406.07  3362.1 2404.82  3482.2 2404.21  3643.1  2401.9  3693.3 2400.09
  3842.6 2398.93  3843.1 2398.92  4190.7 2395.79  4236.3 2396.76  4276.5  2395.5
  4573.9 2395.26    5010 2390.73  5010.5 2390.23  5017.5 2390.73  5536.2 2396.79
  6001.1 2397.34  6044.6  2398.5  6244.7 2397.98  6288.6 2399.25  6484.7 2398.65
  6530.4 2399.72  6560.1 2398.86  6684.9 2399.81  6728.4 2398.74  7067.5 2399.42
#Mann= 6 ,-1 , 0
  2989.5    .035       0  3362.1     .07       0  3842.6    .045       0
  3843.1     .07       0    5010     .07       0  5017.5     .07       0
Bank Sta=5010,5017.5
XS Rating Curve= 0 ,0
Exp/Cntr=0.3,0.1

Type RM Length L Ch R = 1 ,33873   ,439,439,439
BEGIN DESCRIPTION:
Long Branch 65.0
END DESCRIPTION:
XS GIS Cut Line= 3
      1349304.95        6844088.      1351328.11      6844111.73
        1351905.        6842288.
#Sta/Elev= 30
  2976.7 2404.69  3158.5  2402.3  3486.8 2398.66  3506.8 2399.88  3536.8 2397.81
  3756.8  2395.9  3796.8 2396.85  3826.8 2395.38  4036.8 2394.05  4076.8 2395.08
  4106.8 2393.62  4336.8 2391.78  4506.9 2391.64  4576.9 2393.34    4666 2392.28
  4736.9 2393.27    4864 2390.72  4925.9 2391.16  4991.8 2388.37  4992.3 2387.87
    5000 2388.37    5040 2389.14  5087.9 2392.25  5098.3 2391.16  5104.6 2392.27
  5201.6 2391.11  5318.6 2394.26  5637.4 2395.65  5675.2 2396.92  6912.8 2399.53
#Mann= 8 ,-1 , 0
  2976.7     .07       0  3158.5    .045       0    4666    .035       0
    4864     .07       0  4925.9    .035       0  4991.8    .035       0
    5000    .035       0  5087.9     .07       0
Bank Sta=4991.8,5000
XS Rating Curve= 0 ,0
Exp/Cntr=0.3,0.1

Type RM Length L Ch R = 1 ,33434   ,377,377,377
BEGIN DESCRIPTION:
Long Branch 64.0
END DESCRIPTION:
XS GIS Cut Line= 3
      1350005.02      6845937.98      1351624.84      6844408.07
      1352004.99      6842588.05
#Sta/Elev= 30
  2771.9 2402.95  3585.2 2396.36    4328  2395.6  4363.6 2396.52  4540.4 2393.98
  4575.6 2394.93    4597 2393.12  4655.9 2392.08    4682  2392.8  4713.2  2390.7
  4759.7 2390.75  4925.4 2385.12  4925.9 2384.62  4933.7 2385.12  5002.6 2385.34
  5081.8 2388.29  5112.4 2394.11  5120.3 2393.89  5125.4 2391.21  5143.1 2389.46
  5182.2 2389.94  5339.6 2393.07  5490.4    2394  5551.7 2395.61  5684.5 2395.27
  5725.4 2396.54  6532.4 2398.31  6573.3 2399.63    6604 2398.74  6859.3 2399.46
#Mann= 7 ,-1 , 0
  2771.9    .045       0  4655.9    .035       0  4713.2     .07       0
  4925.4     .07       0  4933.7     .07       0  5182.2    .063       0
  5339.6     .07       0
Bank Sta=4925.4,4933.7
XS Rating Curve= 0 ,0
Exp/Cntr=0.3,0.1

Type RM Length L Ch R = 1 ,33057   ,416,416,416
BEGIN DESCRIPTION:
Long Branch 63.0
END DESCRIPTION:
XS GIS Cut Line= 3
      1350555.01      6845837.99      1351788.67      6844721.31
      1352060.64      6844247.52
#Sta/Elev= 30
    3336 2399.08  3357.3 2397.64  3410.4 2397.24  3562.7 2395.85    3704 2395.68
  4284.6 2395.54    4313 2396.56  4341.3 2395.37  4440.7 2395.49  4546.8  2394.1
  4575.2 2395.04  4615.7 2393.04  4645.5 2392.14  4673.9 2392.94  4695.5 2391.12
  4744.8 2391.03  4763.9 2389.58  4872.6 2385.68  4950.3 2380.67  4971.2 2380.55
  4974.5 2379.04    4975 2378.54  4982.8 2379.04  4985.4 2380.75  5037.7 2384.44
  5059.3 2387.98  5080.9 2386.59  5328.2 2393.29  5500.9 2395.88  5546.3 2396.52
#Mann= 7 ,-1 , 0
    3336     .07       0  3410.4    .045       0  4615.7    .035       0
  4763.9     .07       0  4974.5     .07       0  4982.8     .07       0
  5500.9    .063       0
Bank Sta=4974.5,4982.8
XS Rating Curve= 0 ,0
Exp/Cntr=0.3,0.1

Type RM Length L Ch R = 1 ,32641   ,121,121,121
BEGIN DESCRIPTION:
Long Branch 62.1
END DESCRIPTION:
XS GIS Cut Line= 3
      1351718.41      6845255.58      1351938.25      6845021.54
      1352033.61      6844562.13
#Sta/Elev= 30
  4678.9 2392.71  4752.6 2390.93  4759.5 2390.27    4781 2390.01  4865.9 2386.34
  4880.3 2386.06  4936.3 2383.68  4971.9 2381.66  4978.8 2381.69  4986.1 2380.88
    4993 2381.01    4999  2380.1  5004.3  2380.1  5008.7 2379.38  5009.7 2378.87
  5010.2 2378.37  5017.5 2378.37    5018 2378.87  5075.1 2379.18  5108.9  2381.3
  5126.2 2383.31  5197.7 2386.02  5248.7 2387.16  5279.4 2388.38  5299.3 2388.62
    5310 2389.31  5371.3 2390.03  5412.1 2391.62  5454.8 2391.89  5469.2 2392.34
#Mann= 4 ,-1 , 0
  4678.9    .035       0  4880.3    .063       0  5009.7     .03       0
    5018     .03       0
Bank Sta=5009.7,5018
XS Rating Curve= 0 ,0
Exp/Cntr=0.3,0.1

Type RM Length L Ch R = 1 ,32520   ,576,576,576
BEGIN DESCRIPTION:
Long Branch 62.0
END DESCRIPTION:
XS GIS Cut Line= 3
      1351914.89      6845355.77      1352054.97      6845038.08
      1352105.01      6844587.95
#Sta/Elev= 30
  4652.8 2387.06  4689.4 2386.73  4694.9 2385.98  4712.8 2386.31  4736.1 2385.39
  4759.4 2386.03  4764.9    2385  4788.2 2385.08  4793.7 2384.18  4811.5 2384.15
    4817 2383.63  4840.3 2382.77    4858 2382.45    4939  2378.2  4978.2 2376.95
  4993.2 2376.85  4993.7 2376.35    5001 2376.35  5001.5 2376.85  5040.3 2377.74
  5080.6 2381.01  5120.8 2382.79    5136 2383.12    5141 2382.76  5226.5 2386.29
  5231.6 2386.01  5332.1 2388.85  5407.6 2391.52  5412.6  2391.2  5452.9 2392.52
#Mann= 3 ,-1 , 0
  4652.8    .063       0  4993.2     .16       0  5001.5     .16       0
Bank Sta=4993.2,5001.5
XS Rating Curve= 0 ,0
Exp/Cntr=0.3,0.1

Type RM Length L Ch R = 1 ,31944   ,90,90,90
BEGIN DESCRIPTION:
Long Branch 61.0
END DESCRIPTION:
XS GIS Cut Line= 3
      1352654.99      6845287.96      1352615.05      6844988.11
        1352505.        6844638.
#Sta/Elev= 30
  4697.5 2387.37  4727.7  2386.8    4734 2385.58  4739.1 2385.75  4747.9 2384.35
  4812.3 2382.51  4838.7 2380.45  4885.4 2378.08  4890.5 2378.66  4909.3 2378.15
  4958.6 2373.44  4969.8 2371.61  4979.9 2371.07  5037.7  2370.9  5038.2  2370.4
  5045.9  2370.4  5046.4  2370.9  5094.5  2371.5  5136.4 2373.96  5157.4 2376.43
  5188.8 2377.39  5221.2  2377.4  5230.7 2379.32  5248.4 2380.41  5253.6 2379.91
  5272.7 2380.33  5313.2 2385.22  5318.4 2385.22  5356.5 2389.22    5367 2389.79
#Mann= 3 ,-1 , 0
  4697.5     .07       0  5037.7     .07       0  5046.4     .07       0
Bank Sta=5037.7,5046.4
XS Rating Curve= 0 ,0
Exp/Cntr=0.3,0.1

Type RM Length L Ch R = 1 ,31854   ,341,341,341
BEGIN DESCRIPTION:
Long Branch 60.1
END DESCRIPTION:
XS GIS Cut Line= 3
      1352715.94      6845197.69      1352701.95      6844944.68
      1352579.85       6844598.9
#Sta/Elev= 30
  4785.9 2381.62  4805.6 2383.08  4825.6  2382.1  4835.7  2380.1  4875.7 2377.56
  4897.1 2377.66  4955.8 2374.66  4985.9 2372.47  4995.9 2370.93  5015.9 2369.81
  5052.6 2369.48  5053.1 2368.98  5060.8 2368.98  5061.3 2369.48  5173.6 2375.51
  5184.2 2375.24  5192.4 2374.12  5205.5 2374.12  5223.4 2374.19  5228.7 2375.18
  5247.9  2374.7  5254.3 2375.95  5279.7 2375.12  5290.5 2375.62  5310.8 2377.64
  5341.8 2383.59  5353.9 2384.43  5364.5 2386.16  5403.6 2389.05    5406 2389.92
#Mann= 3 ,-1 , 0
  4785.9     .07       0  5052.6     .07       0  5061.3     .07       0
Bank Sta=5052.6,5061.3
XS Rating Curve= 0 ,0
Exp/Cntr=0.3,0.1

Type RM Length L Ch R = 1 ,31513   ,162,162,162
BEGIN DESCRIPTION:
Long Branch 60.0
END DESCRIPTION:
XS GIS Cut Line= 3
      1352905.01      6845337.97      1352999.08      6844930.18
      1352655.02      6844538.02
#Sta/Elev= 30
  4581.5 2390.25  4622.5 2386.33  4725.1 2379.39  4733.7 2377.53  4738.9 2378.02
  4781.6 2372.43  4810.1 2371.28  4920.2  2372.4  5007.3    2366  5007.8  2365.5
    5016    2366  5018.3 2367.01  5040.1 2367.97  5096.1 2368.75  5174.9 2372.11
  5193.3 2370.79  5245.1 2370.72  5252.7 2373.71  5259.3 2372.46  5273.6 2372.61
  5281.2 2375.68  5295.4 2376.83    5359 2380.49  5394.1 2379.76  5401.7 2382.48
  5408.3  2380.4  5436.8 2384.32  5500.4 2385.88    5508 2387.76  5521.7 2388.65
#Mann= 5 ,-1 , 0
  4581.5     .07       0  4810.1    .035       0  5007.3    .035       0
    5016    .035       0  5193.3     .07       0
Bank Sta=5007.3,5016
XS Rating Curve= 0 ,0
Exp/Cntr=0.3,0.1

Type RM Length L Ch R = 1 ,31351   ,179,179,179
BEGIN DESCRIPTION:
Long Branch 59.2
END DESCRIPTION:
XS GIS Cut Line= 3
      1353109.69      6845149.09      1353142.99      6844889.22
      1353116.46      6844632.28
#Sta/Elev= 30
    4738 2373.23  4779.4  2371.8  4789.5 2370.93  4816.9 2369.81    4822    2370
  4870.2 2368.81  4884.6 2368.14  4890.3 2367.69  4896.6 2367.81  4900.6 2367.27
  4950.8 2365.12  4960.9 2363.59  4976.3 2362.54    4977  2360.4  4977.5  2359.9
  4985.2  2359.9  4985.7  2360.4  5003.1 2361.03  5021.3 2362.41  5027.7 2364.65
  5032.7 2365.93  5041.4 2366.91  5071.6 2368.76  5081.6 2368.82  5091.7 2370.18
  5121.6 2370.33  5131.9 2371.18  5202.3 2373.68  5225.6 2375.07  5258.3 2377.85
#Mann= 5 ,-1 , 0
    4738     .07       0  4884.6    .035       0  4900.6     .07       0
    4977     .07       0  4985.7     .07       0
Bank Sta=4977,4985.7
XS Rating Curve= 0 ,0
Exp/Cntr=0.3,0.1

Type RM Length L Ch R = 1 ,31172   ,158,158,158
BEGIN DESCRIPTION:
Long Branch 59.1
END DESCRIPTION:
XS GIS Cut Line= 3
      1353261.57      6845219.79      1353252.53      6844944.04
      1353181.47      6844675.79
#Sta/Elev= 30
  4724.1 2372.76  4745.9  2372.4  4785.9 2370.71  4824.9 2370.19  4872.3 2369.11
    4906 2368.34    4926  2366.8    4936 2365.83    4946 2362.21    4966 2363.22
    4976 2363.18    4986  2359.3  4991.1 2358.65  4991.6 2358.15  4999.4 2358.15
  4999.9 2358.65  5005.5  2362.7  5010.7 2363.43  5026.9 2361.25  5037.3 2363.21
  5050.9 2364.04    5058 2365.12  5099.4 2365.85  5151.1 2368.04  5171.8 2368.32
  5182.1 2369.04  5241.6 2371.26  5246.8 2371.12  5264.9 2372.79  5277.5 2372.69
#Mann= 5 ,-1 , 0
  4724.1     .07       0  4824.9    .035       0  4872.3     .07       0
  4991.1     .07       0  4999.9     .07       0
Bank Sta=4991.1,4999.9
XS Rating Curve= 0 ,0
Exp/Cntr=0.3,0.1

Type RM Length L Ch R = 1 ,31014   ,271,271,271
BEGIN DESCRIPTION:
Long Branch 59.0
END DESCRIPTION:
XS GIS Cut Line= 3
      1353505.01      6845338.03      1353409.72      6844938.43
      1353354.99      6844537.95
#Sta/Elev= 30
  4589.2 2381.01  4640.6 2376.95  4649.8 2376.69    4655 2378.26  4661.2 2376.84
  4681.8 2374.96  4722.9  2372.6  4786.5 2370.26  4794.8 2370.49    4836 2368.34
  4856.5 2368.25  4887.4 2367.03  4954.9 2362.74  4964.3 2362.69  4990.2  2361.7
  4997.1 2360.89  5002.7 2361.18  5006.1 2356.28  5006.6 2355.78  5014.4 2355.78
  5014.9 2356.28  5020.6  2358.9  5030.7 2361.46  5040.8 2361.78    5074 2365.11
  5151.8 2368.99  5343.6 2375.21  5380.2 2377.57    5388 2378.44  5404.2 2380.31
#Mann= 6 ,-1 , 0
  4589.2    .035       0  4964.3     .07       0  5006.1     .07       0
  5014.9     .07       0  5380.2    .035       0    5388    .063       0
Bank Sta=5006.1,5014.9
XS Rating Curve= 0 ,0
Exp/Cntr=0.3,0.1

Type RM Length L Ch R = 1 ,30743   ,106,106,106
BEGIN DESCRIPTION:
Long Branch 58.1
END DESCRIPTION:
XS GIS Cut Line= 3
      1353606.78      6845128.84      1353664.54      6844887.97
      1353623.49      6844654.45
#Sta/Elev= 30
  4752.3 2370.05  4767.3 2369.58  4794.3 2367.71  4809.4 2367.43  4825.1 2366.34
  4845.7  2365.7  4851.4 2364.84  4893.4 2362.34  4898.5 2362.42  4917.7 2358.12
  4935.4 2356.27  4940.5 2356.69  4964.7 2354.67  4965.2 2354.17    4973 2354.17
  4973.5 2354.67  4977.4 2355.31  5002.5 2354.83  5024.9 2356.49  5040.6  2358.1
  5050.7 2359.74  5060.9 2362.21    5071  2363.2  5085.1 2363.89  5091.3 2364.71
  5144.5 2367.14  5152.3 2367.87  5192.9 2368.82  5213.2 2369.99  5237.1 2370.74
#Mann= 4 ,-1 , 0
  4752.3    .035       0  4964.7    .035       0  4973.5    .035       0
  5024.9     .07       0
Bank Sta=4964.7,4973.5
XS Rating Curve= 0 ,0
Exp/Cntr=0.3,0.1

Type RM Length L Ch R = 1 ,30637   ,548,548,548
BEGIN DESCRIPTION:
Long Branch 58.0
END DESCRIPTION:
XS GIS Cut Line= 3
        1353655.        6845188.      1353770.01      6844887.98
        1353705.        6844638.
#Sta/Elev= 30
  4678.7 2373.09  4681.4 2373.09  4688.4 2371.34  4693.7 2371.68  4700.1 2370.36
  4733.6 2369.01  4839.3 2363.65    4850 2363.46  4903.6 2360.29  4912.6 2360.34
  4935.7 2358.63  4947.9 2358.68  4967.3 2356.98  4972.6 2357.01  4978.6 2355.47
  4984.9 2355.05  4985.4 2354.55  4993.2 2354.55  4993.7 2355.05  4997.3  2355.7
    5000 2355.45  5020.6 2357.23  5043.1 2358.37  5051.6 2360.11    5062 2361.37
  5083.7 2363.05    5093 2362.94    5119  2364.4  5247.2 2369.56  5258.3 2369.85
#Mann= 5 ,-1 , 0
  4678.7    .035       0  4733.6     .07       0  4984.9     .07       0
  4993.7     .07       0  5247.2    .035       0
Bank Sta=4984.9,4993.7
XS Rating Curve= 0 ,0
Exp/Cntr=0.3,0.1

Type RM Length L Ch R = 1 ,30089   ,225,225,225
BEGIN DESCRIPTION:
Long Branch 57.0
END DESCRIPTION:
XS GIS Cut Line= 3
        1353955.        6845288.      1354270.21      6844838.51
        1353955.        6844488.
#Sta/Elev= 30
    4451 2368.74  4464.5 2367.41    4509 2365.54  4573.1 2365.38  4586.5 2364.06
  4651.9 2362.73  4767.8 2358.64  4830.6 2358.49  4910.8 2353.32  4929.2 2352.78
  4952.6 2351.93  4982.3  2352.2  4995.4 2351.39  4995.9 2350.89  5004.3 2351.39
  5025.5 2352.61  5077.6 2352.43  5131.7  2353.4  5202.4 2358.09  5280.4 2361.69
  5294.6  2361.5  5301.3 2362.27  5308.8 2360.21  5329.8 2360.61  5336.9 2360.92
    5344 2362.62  5350.7 2361.98  5358.2  2364.9  5443.4 2365.89  5471.4 2368.26
#Mann= 5 ,-1 , 0
    4451    .035       0  4929.2     .07       0  4995.4     .07       0
  5004.3     .07       0  5077.6    .035       0
Bank Sta=4995.4,5004.3
XS Rating Curve= 0 ,0
Exp/Cntr=0.3,0.1

Type RM Length L Ch R = 1 ,29864   ,167,167,167
BEGIN DESCRIPTION:
Long Branch 4353
END DESCRIPTION:
XS GIS Cut Line= 3
       1354430.6      6845102.35      1354495.91      6844837.99
      1354328.17      6844680.49
#Sta/Elev= 30
  4727.7 2356.46    4809 2356.48  4814.6 2355.81  4855.4 2354.74  4866.1 2354.72
  4876.4 2353.85  4886.7 2353.51  4891.9 2352.81  4917.6 2351.79  4948.5 2349.61
  4958.8 2349.51  4989.7 2350.22    5015 2350.11  5021.9 2350.43  5028.7 2348.91
  5031.6 2348.77  5032.1 2348.27    5040 2348.27  5040.5 2348.77  5057.1 2350.46
  5071.2 2350.22  5092.7 2350.77  5135.2 2351.09  5149.3 2351.47  5163.5 2352.39
    5206 2353.31  5212.8 2354.27  5220.2  2354.5    5227  2355.6  5230.1 2355.48
#Mann= 4 ,-1 , 0
  4727.7     .07       0  4855.4    .035       0  5031.6    .035       0
  5040.5    .035       0
#XS Ineff= 2 , 0
         5021.02 2352.47
Permanent Ineff=
       F       F
Bank Sta=5031.6,5040.5
XS Rating Curve= 0 ,0
Exp/Cntr=0.3,0.1

Type RM Length L Ch R = 1 ,29697   ,209,209,209
BEGIN DESCRIPTION:
Long Branch 56.0
END DESCRIPTION:
XS GIS Cut Line= 3
        1354805.      6845287.99      1354661.06      6844846.14
      1354569.14      6844719.97
#Sta/Elev= 30
  4535.3 2358.96  4583.2 2358.24  4598.4  2357.1  4678.9 2354.76  4803.4 2349.54
  4843.8 2349.21  4850.8 2348.43  4892.9 2348.39  4902.3 2347.63  4907.6 2348.46
  4924.4 2347.77  4934.3 2349.11  4939.5 2347.25  4952.3 2346.14  4966.2 2345.16
  4971.4 2345.81  4987.5 2344.49  4991.9 2343.37  4992.4 2342.87  5000.3 2342.87
  5000.8 2343.37  5010.1 2343.75  5017.5 2345.33  5023.7 2345.09  5038.4 2347.82
  5103.3 2350.67  5124.1 2350.72  5146.2 2352.28  5153.5 2351.88  5156.1 2352.35
#Mann= 5 ,-1 , 0
  4535.3    .035       0  4803.4     .07       0  4952.3    .035       0
  4991.9    .035       0  5000.8    .035       0
#XS Ineff= 2 , 0
         4972.59 2348.11 5018.07         2347.96
Permanent Ineff=
       F       F
Bank Sta=4991.9,5000.8
XS Rating Curve= 0 ,0
Exp/Cntr=0.3,0.1

Type RM Length L Ch R = 1 ,29488   ,285,285,285
BEGIN DESCRIPTION:
Long Branch 4354
END DESCRIPTION:
XS GIS Cut Line= 3
      1354890.66      6845204.75      1354855.18      6844887.63
      1354648.79      6844747.26
#Sta/Elev= 30
  4680.9 2356.67  4684.8 2355.95  4689.8 2356.95  4717.9 2353.07    4738 2351.72
  4768.2  2353.3  4788.3 2351.73  4858.8  2352.1  4865.3 2351.83  4870.3 2349.45
  4909.1 2347.57  4919.1 2345.75  4939.3 2344.89  4955.5 2343.11  4969.4    2344
  5007.2 2344.04  5022.2 2344.01  5023.6 2343.02  5024.1 2342.52  5032.8 2343.02
  5049.2 2345.26  5079.1 2345.58  5085.1 2344.57    5109 2343.23    5136 2346.53
  5150.9 2346.87  5165.9 2350.47  5186.9 2348.41  5237.7 2349.99  5249.6 2351.04
#Mann= 3 ,-1 , 0
  4680.9    .035       0  5023.6    .035       0  5032.8    .035       0
Bank Sta=5023.6,5032.8
XS Rating Curve= 0 ,0
Exp/Cntr=0.3,0.1

Type RM Length L Ch R = 1 ,29203   ,122,122,122
BEGIN DESCRIPTION:
Long Branch 55.1
END DESCRIPTION:
XS GIS Cut Line= 3
      1355382.51      6844947.96      1355111.16      6844880.12
      1354729.72      6844775.99
#Sta/Elev= 30
  4720.3  2348.3  4778.2 2348.07  4783.4 2347.65  4860.7 2348.37  4865.8 2347.44
  4923.9  2347.6  4934.2 2348.31  4943.1 2350.07  4948.3 2355.46  4954.8 2353.87
  4975.4 2347.19  4984.4 2345.57  4989.5 2342.53    5000 2342.01  5012.2 2339.47
  5012.7 2338.97  5020.9 2338.97  5021.4 2339.47  5058.2 2340.25    5079 2341.61
  5098.7 2341.64  5138.5 2343.52  5183.4 2344.54  5224.1 2345.17  5252.4 2344.97
  5257.6 2345.59  5286.3 2345.43    5307 2346.18  5366.4 2346.88  5395.4 2347.91
#Mann= 3 ,-1 , 0
  4720.3    .035       0  5012.2    .035       0  5021.4    .035       0
Bank Sta=5012.2,5021.4
XS Rating Curve= 0 ,0
Exp/Cntr=0.3,0.1

Type RM Length L Ch R = 1 ,29081   ,478,478,478
BEGIN DESCRIPTION:
Long Branch 55.0
END DESCRIPTION:
XS GIS Cut Line= 3
      1355572.74      6844869.05      1355198.84      6844795.88
      1354605.03      6844438.02
#Sta/Elev= 30
    4619  2346.9  4697.9  2346.8  4759.6 2344.85    4806 2344.47  4811.1  2343.1
  4840.9 2341.35  4857.5 2341.82  4862.6 2339.84  4891.8 2341.22    4909 2340.59
  4914.1 2337.87  4942.8 2335.86    4961 2335.75  4961.5 2335.25  4970.2 2335.75
  4999.4 2337.36  5016.2 2337.07  5023.5 2337.73  5029.3 2339.73  5060.4 2340.64
  5087.6 2343.71  5109.6 2344.67  5277.8 2345.97  5473.9 2351.43  5547.7 2352.21
  5590.4 2354.16    5606 2355.79    5635  2354.6  5658.3 2355.12  5693.3 2357.44
#Mann= 3 ,-1 , 0
    4619    .035       0    4961    .035       0  4970.2    .035       0
Bank Sta=4961,4970.2
XS Rating Curve= 0 ,0
Exp/Cntr=0.3,0.1

Type RM Length L Ch R = 1 ,28603   ,394,394,394
BEGIN DESCRIPTION:
Long Branch 54.0
END DESCRIPTION:
XS GIS Cut Line= 3
        1355605.        6844838.      1355568.32      6844524.64
      1355405.03      6844388.03
#Sta/Elev= 30
  4684.5 2346.46  4694.6  2345.9  4728.7 2345.07  4775.1 2342.89  4805.3 2341.91
  4875.8 2338.16  4900.3 2337.58    4906 2337.04  4946.3 2335.27  4956.3 2333.78
  4976.5  2331.9  4983.5 2331.61  4988.6 2330.38    5000 2330.16  5002.1  2328.8
  5002.6  2328.3  5010.8  2328.3  5011.3  2328.8  5014.5 2330.12  5028.8 2331.36
  5051.6 2330.89  5063.9 2331.27  5070.5 2330.77  5113.4 2331.16    5135 2332.05
    5142 2332.78  5162.9    2337    5185 2342.85  5199.3 2344.69  5212.9 2345.52
#Mann= 5 ,-1 , 0
  4684.5    .035       0  5002.1    .035       0  5011.3    .035       0
  5051.6     .07       0    5135    .035       0
Bank Sta=5002.1,5011.3
XS Rating Curve= 0 ,0
Exp/Cntr=0.3,0.1

Type RM Length L Ch R = 1 ,28209   ,496,496,496
BEGIN DESCRIPTION:
Long Branch 53.0
END DESCRIPTION:
XS GIS Cut Line= 3
      1355955.01      6844588.04      1355911.45      6844380.25
        1356005.      6844038.01
#Sta/Elev= 30
  4787.7 2341.61  4818.4 2340.96  4862.6  2338.2  4879.7 2336.76  4907.4 2332.63
  4930.8 2330.16  4981.9 2326.13  4998.6 2325.26  5023.1 2324.78  5030.3  2325.2
  5070.6  2324.2  5071.1  2323.7  5079.4  2323.7  5079.9  2324.2  5104.5 2329.33
  5109.7 2328.28  5116.4 2329.35  5144.2  2329.2  5189.1 2326.32  5199.3 2326.63
  5218.5 2329.26  5223.6  2328.9  5230.4 2330.97  5251.1 2331.96  5258.2 2333.24
  5263.3  2333.1  5282.2  2336.9  5292.6 2337.51  5332.4  2342.5  5354.8  2344.1
#Mann= 3 ,-1 , 0
  4787.7    .035       0  5070.6    .035       0  5079.9    .035       0
Bank Sta=5070.6,5079.9
XS Rating Curve= 0 ,0
Exp/Cntr=0.3,0.1

Type RM Length L Ch R = 1 ,27713   ,489,489,489
BEGIN DESCRIPTION:
Long Branch 52.0
END DESCRIPTION:
XS GIS Cut Line= 3
        1356305.      6844338.02      1356314.09      6844187.99
        1356305.      6844088.01
#Sta/Elev= 30
  4849.7 2329.55  4852.2 2329.55  4859.7 2328.48  4869.8 2327.97  4879.8 2327.82
  4889.8 2326.66  4899.8 2325.69  4909.8 2325.65  4928.6 2325.17  4933.6 2324.39
  4949.9 2323.37  4959.9 2320.76  4969.9 2317.68    4980 2313.63  4985.2 2310.84
  4985.7 2310.34  4994.3 2310.34  4994.8 2310.84  4997.5 2313.16  5002.5 2313.16
    5010 2313.61  5020.1 2315.79  5030.1 2324.01  5040.2 2324.41  5050.2 2325.88
  5080.3 2328.39  5090.4  2328.9  5096.3  2329.4  5097.9 2329.54  5100.4 2329.54
#Mann= 4 ,-1 , 0
  4849.7     .07       0  4985.2     .07       0  4994.8     .07       0
  5096.3    .035       0
Bank Sta=4985.2,4994.8
XS Rating Curve= 0 ,0
Exp/Cntr=0.3,0.1

Type RM Length L Ch R = 1 ,27224   ,498,498,498
BEGIN DESCRIPTION:
Long Branch 51.0
END DESCRIPTION:
XS GIS Cut Line= 3
      1356804.99      6844387.98      1356764.69      6844277.82
      1356555.02      6843888.03
#Sta/Elev= 30
  4882.7 2330.37  4914.6  2323.7  4923.1  2320.3  4928.5 2319.67  4935.9 2316.69
  4958.8 2310.75  4984.2 2303.09  4989.5 2303.96  4992.1 2302.94  4992.6 2302.44
  5002.3 2302.94  5035.3 2306.13  5045.2 2308.24  5051.5 2311.92  5057.2 2310.88
  5073.4 2314.04  5117.2 2315.79  5133.5 2314.82  5155.4  2315.3  5177.3    2317
    5183  2318.3  5199.2 2318.31  5249.6 2321.76  5259.2 2321.31  5281.2  2322.6
  5308.7 2325.31  5340.4 2326.42  5374.5 2330.03    5396 2330.81  5442.6 2337.89
#Mann= 5 ,-1 , 0
  4882.7    .035       0  4958.8     .07       0  4992.1     .07       0
  5002.3     .07       0    5396    .035       0
Bank Sta=4992.1,5002.3
XS Rating Curve= 0 ,0
Exp/Cntr=0.3,0.1
