HEC-RAS study Long Branch.prj: Long Branch Base Level Engineering

--- Long Branch.g01 (geometry) --- (continued)

Type RM Length L Ch R = 1 ,26726   ,278,278,278
BEGIN DESCRIPTION:
Long Branch 50.0
END DESCRIPTION:
XS GIS Cut Line= 3
        1357055.      6844187.98      1357085.32      6843958.38
      1357055.01      6843838.03
#Sta/Elev= 30
  4768.4 2320.72  4770.9 2320.72  4788.6 2317.64  4805.1 2313.09  4810.2 2313.29
  4828.9  2310.5    4839  2309.8  4859.2 2307.23  4889.4 2305.38  4970.1 2302.93
  4980.2 2301.66  4990.3 2299.59  4997.7 2296.41  5002.8 2296.41  5005.5 2294.28
    5006 2293.78  5015.3 2293.78  5015.8 2294.28  5031.3 2296.15  5051.9 2300.94
  5059.9 2303.66  5065.1 2303.24  5072.6 2305.74  5082.9  2306.4  5093.2 2308.16
    5101 2313.08  5106.2 2315.56  5113.8 2317.05  5121.6 2320.12  5124.1 2320.12
#Mann= 3 ,-1 , 0
  4768.4     .07       0  5005.5     .07       0  5015.8     .07       0
Bank Sta=5005.5,5015.8
XS Rating Curve= 0 ,0
Exp/Cntr=0.3,0.1

Type RM Length L Ch R = 1 ,26448   ,218,218,218
BEGIN DESCRIPTION:
Long Branch 4239
END DESCRIPTION:
XS GIS Cut Line= 3
      1357233.41      6844230.78      1357315.01      6843887.96
      1357216.67      6843742.11
#Sta/Elev= 30
  4647.6 2311.56  4681.3 2309.71  4732.7 2308.34  4753.2    2307  4794.4 2307.11
  4849.8 2305.26  4886.9 2301.73    4892 2302.38  4897.2 2300.67  4917.7 2297.59
    4928 2298.06  4939.3 2296.73  4958.8 2296.88  4984.5 2292.84    4985 2292.34
  4994.3 2292.34  4994.8 2292.84    5003 2293.17  5007.5 2294.98  5013.5 2294.66
  5028.5 2297.38  5036.1 2301.63  5058.4 2305.35  5064.5 2305.62  5094.4 2313.68
  5100.4 2314.64  5108.5 2319.11  5115.4 2322.07  5151.4 2325.16  5175.9 2326.03
#Mann= 3 ,-1 , 0
  4647.6     .07       0  4984.5     .07       0  4994.8     .07       0
Bank Sta=4984.5,4994.8
XS Rating Curve= 0 ,0
Exp/Cntr=0.3,0.1

Type RM Length L Ch R = 1 ,26230   ,179,179,179
BEGIN DESCRIPTION:
Long Branch 4238
END DESCRIPTION:
XS GIS Cut Line= 3
      1357412.25      6844163.03      1357511.73      6843944.51
      1357478.21      6843765.52
#Sta/Elev= 30
  4759.9 2310.17  4774.8 2308.69  4864.3 2303.36  4886.3 2301.53  4895.5 2299.87
    4901 2299.81  4908.3 2297.25  4930.2 2293.15  4947.1 2291.41  4970.2 2293.07
  4985.2  2293.1    5000 2291.38  5000.3 2290.35  5000.8 2289.85  5010.1 2289.85
  5010.6 2290.35    5027 2292.65  5037.1 2296.02  5057.5 2296.95  5063.2 2298.01
  5068.2  2297.6  5077.8 2298.15    5088 2301.33  5108.4  2309.5  5115.8 2314.68
  5120.8  2314.4  5128.7 2318.64  5138.9 2321.49  5159.2 2323.84  5182.1 2325.62
#Mann= 3 ,-1 , 0
  4759.9     .07       0  5000.3     .07       0  5010.6     .07       0
Bank Sta=5000.3,5010.6
XS Rating Curve= 0 ,0
Exp/Cntr=0.3,0.1

Type RM Length L Ch R = 1 ,26051   ,285,285,285
BEGIN DESCRIPTION:
Long Branch 49.0
END DESCRIPTION:
XS GIS Cut Line= 3
        1357655.        6844188.      1357653.35       6844034.9
      1357540.72      6843788.09
#Sta/Elev= 30
  4846.9 2321.13  4866.9 2317.46  4876.9 2314.19  4886.9 2309.63  4896.9 2303.63
  4906.9  2299.5  4956.9  2294.5  4966.9 2292.52  4973.4 2289.08  4976.9 2287.22
  4999.9 2286.19  5000.4 2285.69  5010.3 2286.19  5010.6 2287.14  5033.6 2288.68
  5051.2 2291.82  5056.7 2291.77  5062.6 2293.99  5079.7 2296.76  5085.2 2296.44
  5102.7 2297.96  5117.5 2298.11  5161.5 2303.18  5171.8 2303.22  5194.5 2305.47
  5223.4 2309.92  5228.9 2311.59  5246.4 2313.42  5251.9 2315.11  5271.3 2316.74
#Mann= 4 ,-1 , 0
  4846.9    .035       0  4973.4     .07       0  4999.9     .07       0
  5010.3     .07       0
Bank Sta=4999.9,5010.3
XS Rating Curve= 0 ,0
Exp/Cntr=0.3,0.1

Type RM Length L Ch R = 1 ,25766   ,499,499,499
BEGIN DESCRIPTION:
Long Branch 48.0
END DESCRIPTION:
XS GIS Cut Line= 3
        1357855.        6843988.      1357824.71      6843817.88
      1357454.96      6843687.98
#Sta/Elev= 30
  4827.2 2310.15  4864.9 2303.97  4898.3 2298.32  4913.1 2288.18  4959.2  2286.5
  4984.5 2281.18    4985 2280.68  4994.9 2281.18  5015.2 2281.89  5020.9 2286.15
  5031.5 2289.64  5045.8 2289.15  5063.3  2291.5  5077.1  2290.3    5095  2291.8
  5116.3 2291.73  5170.1 2296.76  5190.5  2301.1  5195.8 2300.25  5201.1 2303.06
  5221.4 2307.75  5226.7 2306.35  5232.9 2309.16  5252.4 2313.26  5257.7 2312.48
  5283.4 2318.93  5288.7 2317.64  5345.4 2326.64  5350.7  2325.5  5391.9 2328.86
#Mann= 6 ,-1 , 0
  4827.2    .035       0  4864.9     .07       0  4984.5     .07       0
  4994.9     .07       0  5045.8     .16       0    5095     .07       0
Bank Sta=4984.5,4994.9
XS Rating Curve= 0 ,0
Exp/Cntr=0.3,0.1

Type RM Length L Ch R = 1 ,25267   ,498,498,498
BEGIN DESCRIPTION:
Long Branch 47.0
END DESCRIPTION:
XS GIS Cut Line= 3
        1358205.      6844037.98      1358203.86      6843528.58
        1358105.        6843288.
#Sta/Elev= 30
  4490.6 2324.96  4540.6 2319.72  4580.6 2310.42  4590.6 2308.98  4600.6 2306.08
  4620.6 2303.08  4670.6 2298.35  4720.6 2295.19  4790.6 2292.27  4920.6 2289.73
  4940.6 2281.74  4950.6 2280.53  4960.6 2281.27  5015.5  2279.9    5016  2279.4
  5029.1  2279.9  5095.6 2280.18  5120.2 2280.54  5130.4 2281.94  5144.1 2285.96
    5152 2287.19  5162.7 2287.37  5173.6 2289.86  5184.4 2295.12  5192.1 2300.51
    5216  2313.3  5221.4 2316.71  5227.7 2322.96  5238.5 2325.21  5260.1  2327.3
#Mann= 4 ,-1 , 0
  4490.6     .07       0  5015.5     .07       0  5029.1     .07       0
  5095.6     .07       0
Bank Sta=5015.5,5029.1
XS Rating Curve= 0 ,0
Exp/Cntr=0.3,0.1

Type RM Length L Ch R = 1 ,24769   ,491,491,491
BEGIN DESCRIPTION:
Long Branch 46.0
END DESCRIPTION:
XS GIS Cut Line= 3
        1358305.      6843987.99      1358486.73      6843488.21
        1358455.      6843288.01
#Sta/Elev= 30
  4468.2 2321.84  4500.1 2318.41  4539.4 2308.18  4569.9 2301.87  4600.5 2297.59
  4606.5 2295.29  4734.2 2290.36  4809.4 2285.54  4819.3 2285.98  4865.2 2280.76
  4890.5 2279.46  4957.5 2279.07  4982.3 2278.34  4989.6 2276.81  4997.4 2272.98
  5002.6 2272.98  5003.5 2271.22    5004 2270.72  5017.1 2271.22  5039.3 2276.95
  5050.8 2278.46  5058.6 2281.96  5091.3 2301.97  5101.5 2304.83  5111.8  2309.9
  5131.8 2310.29    5169 2318.63  5174.1 2318.29  5182.5 2320.38  5202.7 2322.23
#Mann= 5 ,-1 , 0
  4468.2     .07       0  4957.5     .16       0  5003.5     .07       0
  5017.1     .16       0  5058.6     .07       0
Bank Sta=5003.5,5017.1
XS Rating Curve= 0 ,0
Exp/Cntr=0.3,0.1

Type RM Length L Ch R = 1 ,24278   ,463,463,463
BEGIN DESCRIPTION:
Long Branch 45.0
END DESCRIPTION:
XS GIS Cut Line= 3
        1358905.        6844238.       1358905.1       6843637.9
      1358804.98      6843437.97
#Sta/Elev= 30
  4399.9 2325.38  4479.9 2315.64  4529.9 2306.14  4569.9 2299.83  4579.9 2297.21
  4645.8 2291.49  4779.9 2277.22  4799.9 2276.04  4829.9 2276.43  4849.9 2273.09
  4859.9 2272.54  4879.9 2276.86  4919.9 2276.12  4959.9 2274.13  4989.9 2271.37
    5000 2269.54  5001.6 2268.36  5002.1 2267.86  5015.2 2268.36  5022.3 2268.74
  5030.8 2273.56  5036.4 2273.86  5053.1 2284.82  5058.7 2282.95  5075.5 2288.44
  5081.1 2287.64  5097.8 2290.99  5111.7 2292.51  5187.2 2307.07  5223.6 2310.98
#Mann= 4 ,-1 , 0
  4399.9    .035       0  4645.8     .07       0  5001.6     .07       0
  5015.2     .07       0
Bank Sta=5001.6,5015.2
XS Rating Curve= 0 ,0
Exp/Cntr=0.3,0.1

Type RM Length L Ch R = 1 ,23815   ,498,498,498
BEGIN DESCRIPTION:
Long Branch 44.0
END DESCRIPTION:
XS GIS Cut Line= 3
      1359654.99        6843838.      1359303.28      6843683.86
      1359104.97      6843437.96
#Sta/Elev= 30
    4616 2315.64  4624.9 2314.19  4653.8 2303.79  4659.7 2299.86  4670.6 2296.12
  4677.2 2291.97  4700.5 2281.91  4714.3 2279.78  4781.6 2275.02  4822.9 2274.22
  4875.1 2270.06  4880.5 2271.17  4888.9 2269.99  4921.7 2269.84  4927.3 2267.72
  4932.7 2267.37  4979.5 2267.18  4995.9 2265.99  4996.4 2265.49  5010.5 2265.99
  5017.6 2269.18  5073.6 2273.97  5081.5 2276.46  5095.9 2278.28  5116.7 2279.79
  5137.5 2279.72  5223.9 2285.91  5238.3 2288.25  5279.9 2298.84  5315.9 2306.16
#Mann= 3 ,-1 , 0
    4616     .07       0  4995.9     .07       0  5010.5     .07       0
Bank Sta=4995.9,5010.5
XS Rating Curve= 0 ,0
Exp/Cntr=0.3,0.1

Type RM Length L Ch R = 1 ,23317   ,496,496,496
BEGIN DESCRIPTION:
Long Branch 43.0
END DESCRIPTION:
XS GIS Cut Line= 3
      1359705.02      6843538.04      1359610.81      6843335.69
      1359105.01        6843388.
#Sta/Elev= 30
  4776.8  2293.4  4808.4 2290.82  4831.3  2285.8  4898.2 2278.85  4910.9 2271.97
  4920.2 2270.49  4928.3 2270.87  4933.8 2266.81  4951.2 2265.21  4956.7 2261.71
  4964.4 2260.17  4979.6 2257.79    5000  2258.2  5008.5 2257.01    5009 2256.51
  5023.2 2257.01  5039.3 2261.29  5056.1 2264.82  5071.1 2265.57  5076.2 2267.39
  5096.3 2266.11  5136.5 2267.24  5176.7 2270.98  5263.8 2276.28  5397.9 2282.56
    5418 2285.17  5428.1 2287.86  5478.3 2304.08  5488.4 2306.08  5508.5 2307.41
#Mann= 4 ,-1 , 0
  4776.8     .07       0  5008.5     .07       0  5023.2     .07       0
  5039.3     .07       0
Bank Sta=5008.5,5023.2
XS Rating Curve= 0 ,0
Exp/Cntr=0.3,0.1

Type RM Length L Ch R = 1 ,22821   ,474,474,474
BEGIN DESCRIPTION:
Long Branch 42.0
END DESCRIPTION:
XS GIS Cut Line= 3
      1359955.02      6843238.02      1359654.91      6842882.96
      1359455.01      6842788.01
#Sta/Elev= 30
  4535.1 2286.01  4648.9 2276.39    4762 2272.31  4882.9 2269.74  4897.2 2268.37
  4903.7 2265.93  4911.5 2265.89    4918 2263.53  4932.3 2261.28  4975.2 2258.65
  4981.7 2256.56  5003.6 2255.02  5004.1 2254.52  5018.4 2255.02  5019.9 2257.81
  5025.4 2257.39  5033.1 2260.55  5042.6 2261.86  5048.1 2261.15  5065.3 2263.34
  5070.8 2262.57    5088  2264.3  5093.6 2262.94  5099.5 2264.72  5144.5 2267.81
  5154.9 2271.35  5161.7 2275.07  5167.3 2273.55    5177 2277.52  5221.3 2283.18
#Mann= 3 ,-1 , 0
  4535.1     .07       0  5003.6     .07       0  5018.4     .07       0
Bank Sta=5003.6,5018.4
XS Rating Curve= 0 ,0
Exp/Cntr=0.3,0.1

Type RM Length L Ch R = 1 ,22347   ,481,481,481
BEGIN DESCRIPTION:
Long Branch 41.0
END DESCRIPTION:
XS GIS Cut Line= 3
      1360005.01      6843088.03       1359824.9      6842467.03
      1359904.99      6842238.03
#Sta/Elev= 30
  4353.4 2274.57  4403.8 2272.05    4468 2271.12  4587.2 2267.56  4603.3  2265.7
    4626 2265.89  4726.7 2260.59  4811.6    2260  4837.8 2257.97    4843 2258.55
  4871.4 2255.82  4967.7 2255.15  4977.3 2254.69  4989.3 2251.68  4989.8 2251.18
  5004.5 2251.68  5015.2 2253.78  5020.5 2252.54  5046.2 2260.14  5051.9 2265.32
  5062.5 2270.78  5077.2 2274.47  5083.7 2278.87    5103 2284.42  5108.3 2291.53
  5126.1 2291.44  5147.3 2292.81  5189.7 2291.89  5210.8 2294.25  5242.6 2295.95
#Mann= 3 ,-1 , 0
  4353.4     .07       0  4989.3     .07       0  5004.5     .07       0
Bank Sta=4989.3,5004.5
XS Rating Curve= 0 ,0
Exp/Cntr=0.3,0.1

Type RM Length L Ch R = 1 ,21866   ,498,498,498
BEGIN DESCRIPTION:
Long Branch 40.0
END DESCRIPTION:
XS GIS Cut Line= 3
      1360104.99      6842738.01      1360252.69      6842493.68
      1360304.99      6842288.03
#Sta/Elev= 30
  4714.5 2268.17    4765  2265.7  4817.3 2258.86  4889.8 2257.23    4904 2254.45
  4912.4 2251.74  4918.2 2255.08  4933.7 2248.26  4939.6 2249.88  4948.2 2246.72
  4956.7 2246.58  4968.8 2246.01  4969.3 2245.51    4984 2246.01    4992  2249.5
  4997.4 2246.25  5007.4  2248.3  5025.5 2252.43  5071.6 2252.81  5078.1 2254.71
  5098.7 2261.14  5107.3 2266.19  5112.5 2265.43  5148.3 2290.08  5153.4 2288.97
  5160.6 2295.68  5165.8 2297.66  5189.2 2305.52  5194.3 2304.83  5212.2 2308.51
#Mann= 7 ,-1 , 0
  4714.5     .07       0    4904     .16       0  4956.7     .07       0
  4968.8     .07       0    4984     .07       0  5007.4     .16       0
  5165.8     .07       0
Bank Sta=4968.8,4984
XS Rating Curve= 0 ,0
Exp/Cntr=0.3,0.1

Type RM Length L Ch R = 1 ,21368   ,493,493,493
BEGIN DESCRIPTION:
Long Branch 39.0
END DESCRIPTION:
XS GIS Cut Line= 3
        1360455.      6843288.01      1360655.15       6842687.7
        1360555.      6842387.99
#Sta/Elev= 30
  4367.2 2280.87  4414.6 2275.12  4430.5 2268.96  4451.5 2267.04  4767.8 2258.79
  4888.9 2259.47  4920.6 2257.23  4946.9 2249.39  4952.2 2250.93  4957.5 2247.93
  4987.9 2245.75  4989.6 2243.63  4990.1 2243.13  5004.8 2243.63  5041.9 2245.93
  5047.5 2248.62  5073.5 2250.77  5079.1 2253.67  5157.8 2254.29    5200 2259.63
  5205.4 2262.35  5210.7 2261.83  5231.6 2268.17    5237 2272.07  5263.3 2283.44
  5268.6  2290.1  5273.9 2289.16  5290.3 2296.69  5300.2 2303.06    5316 2304.44
#Mann= 5 ,-1 , 0
  4367.2     .07       0  4987.9     .16       0  4989.6     .07       0
  5004.8     .16       0  5290.3     .07       0
Bank Sta=4989.6,5004.8
XS Rating Curve= 0 ,0
Exp/Cntr=0.3,0.1

Type RM Length L Ch R = 1 ,20875   ,997,997,997
BEGIN DESCRIPTION:
Long Branch 38.0
END DESCRIPTION:
XS GIS Cut Line= 3
      1360905.01      6843287.97      1361091.93      6842673.89
      1361155.01      6842387.96
#Sta/Elev= 30
  4358.1 2268.59  4452.1 2262.04  4576.8 2257.93    4588 2256.14    4653 2253.32
  4718.7 2252.39  4751.5 2249.46  4828.5 2248.63    4921 2251.01  4964.3 2250.13
  4985.2 2244.33  5008.6 2243.46  5009.1 2242.96  5023.9 2243.46  5026.5  2246.4
    5047 2246.26  5077.7 2249.16  5083.4 2251.19  5088.5 2254.83  5098.2 2257.75
    5127 2261.89  5132.2 2264.56  5149.4 2268.88    5181 2280.22  5208.9 2280.86
  5224.7 2282.22  5241.6 2288.36    5262 2298.04  5268.4 2305.59  5292.8 2311.02
#Mann= 4 ,-1 , 0
  4358.1     .07       0  5008.6     .07       0  5023.9     .07       0
  5208.9     .07       0
Bank Sta=5008.6,5023.9
XS Rating Curve= 0 ,0
Exp/Cntr=0.3,0.1

Type RM Length L Ch R = 1 ,19878   ,419,419,419
BEGIN DESCRIPTION:
Long Branch 37.0
END DESCRIPTION:
XS GIS Cut Line= 3
        1361605.      6843137.97      1361635.08      6842808.03
      1361305.02      6842288.04
#Sta/Elev= 30
  4668.7    2262  4723.8 2260.92    4759 2257.25  4814.2 2257.46  4834.1 2258.14
  4859.5 2256.94  4869.5 2255.86  4899.6 2247.84  4929.7 2245.65  4939.4 2246.32
  4944.4  2251.7    4980 2239.63  5027.9 2238.28  5028.4 2237.78  5043.3 2238.28
  5086.5 2243.76  5180.5 2241.92  5253.4 2249.02    5311 2252.26  5341.5 2256.52
  5347.4 2258.68  5362.7 2259.14  5368.6 2261.34  5420.3 2264.57  5450.1 2269.92
  5477.9 2281.37  5535.5 2290.83  5550.7 2294.44  5593.1 2308.69  5615.9 2312.71
#Mann= 4 ,-1 , 0
  4668.7    .035       0  4814.2     .07       0  5027.9     .07       0
  5043.3     .07       0
Bank Sta=5027.9,5043.3
XS Rating Curve= 0 ,0
Exp/Cntr=0.3,0.1

Type RM Length L Ch R = 1 ,19459   ,497,497,497
BEGIN DESCRIPTION:
Long Branch 36.0
END DESCRIPTION:
XS GIS Cut Line= 3
      1362204.98      6843037.97      1361721.43      6842421.23
      1361554.99      6842287.99
#Sta/Elev= 30
  4216.3 2259.27  4387.1 2246.04  4451.3 2246.33  4472.1 2242.15  4494.7 2240.09
  4529.9 2241.04  4544.4 2244.49  4550.8 2249.06  4558.9 2249.67  4565.2 2252.42
  4579.7 2251.17  4629.4  2251.6  4672.8 2249.57  4679.1 2248.22  4728.8 2247.14
  4836.4 2247.35  4871.7 2241.29  4971.1 2236.66  4991.1 2229.98  4991.6 2229.48
  5006.6 2229.98  5013.9 2236.85  5034.7  2243.5  5042.7 2248.24  5085.1 2256.98
  5121.2 2259.89  5170.8 2267.62  5185.2 2271.98    5210 2283.64  5213.2 2283.64
#Mann= 3 ,-1 , 0
  4216.3     .07       0  4991.1     .07       0  5006.6     .07       0
Bank Sta=4991.1,5006.6
XS Rating Curve= 0 ,0
Exp/Cntr=0.3,0.1

Type RM Length L Ch R = 1 ,18962   ,486,486,486
BEGIN DESCRIPTION:
Long Branch 35.0
END DESCRIPTION:
XS GIS Cut Line= 3
      1362355.02      6842788.05      1362138.44      6842204.86
      1362204.99      6841988.05
#Sta/Elev= 30
  4377.9 2252.96  4503.9 2248.54  4509.2  2246.2  4516.6  2245.5  4542.4 2246.93
  4580.6 2243.43    4602 2237.59    4666 2233.21    4698 2232.56  4761.2 2237.22
  4882.6 2238.25    4922 2233.67  4968.4 2231.92  4985.7 2227.65  4986.2 2227.15
  5001.2 2227.65  5003.6 2231.01  5036.4 2232.32  5041.6 2236.09  5059.5 2237.92
  5090.9 2247.18  5107.1  2247.6  5122.2 2253.82  5164.1 2263.98  5172.5 2267.47
    5185 2275.83  5205.3 2282.78  5216.4 2290.78  5224.2 2294.73  5226.8 2294.73
#Mann= 4 ,-1 , 0
  4377.9    .035       0  4542.4     .07       0  4985.7     .07       0
  5001.2     .07       0
Bank Sta=4985.7,5001.2
XS Rating Curve= 0 ,0
Exp/Cntr=0.3,0.1

Type RM Length L Ch R = 1 ,18476   ,401,401,401
BEGIN DESCRIPTION:
Long Branch 34.0
END DESCRIPTION:
XS GIS Cut Line= 3
      1362548.84      6842779.46      1362517.98      6842387.58
      1362304.99      6841937.97
#Sta/Elev= 30
  4606.9 2250.96  4738.8 2246.72  4768.9 2243.46    4819 2241.24  4839.1 2236.96
  4859.1 2237.97  4909.3 2232.38  4959.5 2230.17  4974.4 2225.15  4989.3 2223.65
  4989.8 2223.15  5005.3 2223.65  5010.6 2225.83  5017.4 2232.11  5022.9 2227.33
  5045.7 2232.61  5099.1 2234.78  5113.9 2239.45  5159.4 2240.69  5182.1 2243.85
  5324.1  2255.3  5369.6 2261.71  5397.9 2271.27  5415.1 2281.32  5420.6 2281.48
  5431.1 2286.17  5437.8 2294.09  5443.4 2293.74  5453.2 2298.06  5497.5 2305.53
#Mann= 3 ,-1 , 0
  4606.9     .07       0  4989.3     .07       0  5005.3     .07       0
Bank Sta=4989.3,5005.3
XS Rating Curve= 0 ,0
Exp/Cntr=0.3,0.1

Type RM Length L Ch R = 1 ,18075   ,653,653,653
BEGIN DESCRIPTION:
Long Branch 33.0
END DESCRIPTION:
XS GIS Cut Line= 3
      1363455.02      6842988.02       1362876.1      6842468.41
      1362354.98      6841937.98
#Sta/Elev= 30
  4222.1 2295.85  4250.2 2287.59    4286 2280.53  4413.1 2265.43  4490.9 2250.37
  4611.8 2239.95  4639.6 2233.08  4675.5 2237.96  4795.6  2240.4    4827  2238.7
  4958.8 2231.99    4973 2227.72  4979.2 2222.98  4979.7 2222.48  4995.3 2222.98
  4997.4 2228.04    5033 2228.52  5050.6 2226.69  5071.7 2229.78    5216 2228.84
  5262.7 2229.08    5291 2238.36  5595.1 2257.21  5637.5 2265.63  5665.8 2276.15
  5679.9 2286.22  5701.2    2295  5708.2 2295.77  5715.3  2299.6  5743.6 2303.75
#Mann= 7 ,-1 , 0
  4222.1     .07       0  4795.6    .035       0    4827     .07       0
  4979.2     .07       0  4995.3     .07       0    5033     .16       0
    5216     .07       0
Bank Sta=4979.2,4995.3
XS Rating Curve= 0 ,0
Exp/Cntr=0.3,0.1

Type RM Length L Ch R = 1 ,17422   ,433,433,433
BEGIN DESCRIPTION:
Long Branch 32.0
END DESCRIPTION:
XS GIS Cut Line= 3
      1363505.02      6842838.04       1363221.8      6842221.58
      1362805.01      6841738.01
#Sta/Elev= 30
  4321.6 2271.97  4404.8 2258.64  4464.7 2253.99  4640.1 2244.95  4840.5 2240.32
    4858 2236.71  4863.5 2238.15  4932.4 2230.88  4970.3 2216.56  4970.8 2216.06
  4986.5 2216.56  4992.9 2224.78  4999.2 2225.35    5029 2225.83  5064.1 2229.68
  5184.8 2231.63  5227.5 2234.76  5276.9 2234.65  5397.6 2245.17  5404.2 2244.73
  5482.1 2253.76    5504 2258.85  5510.6 2263.23  5532.5 2270.35    5546 2278.24
  5553.4 2280.28  5581.9  2296.3  5588.5 2301.28    5617 2312.56  5638.4 2317.06
#Mann= 3 ,-1 , 0
  4321.6     .07       0  4970.3     .07       0  4986.5     .07       0
Bank Sta=4970.3,4986.5
XS Rating Curve= 0 ,0
Exp/Cntr=0.3,0.1

Type RM Length L Ch R = 1 ,16989   ,500,500,500
BEGIN DESCRIPTION:
Long Branch 31.0
END DESCRIPTION:
XS GIS Cut Line= 3
      1363511.89      6842404.22      1363454.35      6841872.72
      1363209.68       6841488.4
#Sta/Elev= 30
  4465.4 2240.19  4793.5 2235.61  4923.2 2229.94  4984.6 2220.93  4994.7 2221.53
    5004 2219.46  5009.3 2214.72  5009.8 2214.22  5025.6 2214.72    5031 2218.66
    5053 2222.57  5131.8 2224.74  5183.4    2229  5228.2 2239.78  5270.6 2243.09
  5291.7 2247.26  5343.4 2264.14  5349.4 2270.67  5358.6 2275.59  5364.5 2275.12
  5373.1 2279.81  5379.8 2287.37  5385.7 2285.53    5395  2291.6  5400.9 2290.99
  5416.2 2304.06  5422.1  2302.1  5431.4 2306.45  5437.3 2304.95  5455.6 2310.09
#Mann= 5 ,-1 , 0
  4465.4     .07       0  4923.2     .16       0  5009.3     .07       0
  5025.6     .16       0  5131.8     .07       0
Bank Sta=5009.3,5025.6
XS Rating Curve= 0 ,0
Exp/Cntr=0.3,0.1

Type RM Length L Ch R = 1 ,16489   ,493,493,493
BEGIN DESCRIPTION:
Long Branch 30.0
END DESCRIPTION:
XS GIS Cut Line= 3
      1363554.99      6842388.01      1363799.84      6841888.38
      1363404.99      6841287.98
#Sta/Elev= 30
  4443.6 2239.47  4677.1 2233.56  4778.2 2226.03  4913.2 2223.19  4930.1 2218.19
  4935.7  2220.2  4952.6 2212.85  4958.2 2214.08  4958.9 2211.55  4959.4 2211.05
  4975.2 2211.55  4989.3 2219.04  5120.1  2219.9  5162.8 2224.23  5227.9 2223.99
  5242.9 2226.17  5271.2 2227.98  5277.2 2232.59  5292.3 2235.99  5407.4 2249.79
  5467.1 2258.81  5473.1 2262.13  5488.1 2258.85  5494.1 2263.45  5503.1 2263.68
  5551.3 2277.06  5638.7 2289.65    5690 2292.86  5717.5 2299.24  5718.6 2299.24
#Mann= 5 ,-1 , 0
  4443.6     .07       0  4958.9     .07       0  4975.2     .07       0
  5242.9     .07       0  5717.5    .035       0
Bank Sta=4958.9,4975.2
XS Rating Curve= 0 ,0
Exp/Cntr=0.3,0.1

Type RM Length L Ch R = 1 ,15996   ,492,492,492
BEGIN DESCRIPTION:
Long Branch 29.0
END DESCRIPTION:
XS GIS Cut Line= 3
        1364155.      6842337.98       1364181.3      6842114.82
      1364255.01      6841837.97
#Sta/Elev= 30
  4775.3  2228.7  4825.6 2228.13    4876  2226.1  4896.1 2223.28  4916.2 2217.09
  4946.5 2214.61  4956.5 2211.38  4965.3 2215.07  4966.6 2215.62  4976.7 2213.15
  4982.1 2207.57  4982.6 2207.07  4998.1 2207.07  4998.6 2207.57    5000  2207.8
  5007.1 2211.86  5017.4 2215.43  5027.8 2216.42  5033.4 2217.74  5038.6 2217.52
  5048.5 2219.88  5058.8 2220.78  5068.3 2219.97  5089.8 2219.69  5148.6 2221.01
  5162.3 2220.64  5195.9 2222.23  5245.1 2224.65    5269 2226.87  5286.5    2230
#Mann= 5 ,-1 , 0
  4775.3     .07       0  4965.3     .16       0  4982.1     .07       0
  4998.6     .16       0  5195.9     .07       0
Bank Sta=4982.1,4998.6
XS Rating Curve= 0 ,0
Exp/Cntr=0.3,0.1

Type RM Length L Ch R = 1 ,15504   ,498,498,498
BEGIN DESCRIPTION:
Long Branch 28.0
END DESCRIPTION:
XS GIS Cut Line= 3
      1364636.58      6842820.08      1364607.29      6842182.15
        1364405.        6841888.
#Sta/Elev= 30
  4361.4 2241.06  4423.5 2237.73  4433.6 2238.18  4506.7 2232.52  4543.7 2231.78
  4603.7 2227.18  4673.8  2223.8  4693.8 2221.47    4756 2219.67  4803.9 2217.88
    4824 2215.52    4844 2216.67    4864 2216.14    4874 2217.16    4894 2213.85
  4924.1 2212.27  4974.1 2212.82  4984.1 2211.89  4991.3 2204.62  4991.8 2204.12
  5007.9 2204.62    5012 2207.48  5026.9 2213.15  5140.5 2212.44  5155.4 2214.72
  5170.3 2219.08  5176.4 2222.13  5191.3 2224.41  5304.7 2226.06    5357 2227.31
#Mann= 5 ,-1 , 0
  4361.4     .07       0    4756     .16       0  4991.3     .07       0
  5007.9     .16       0  5304.7     .07       0
Bank Sta=4991.3,5007.9
XS Rating Curve= 0 ,0
Exp/Cntr=0.3,0.1

Type RM Length L Ch R = 1 ,15006   ,498,498,498
BEGIN DESCRIPTION:
Long Branch 27.0
END DESCRIPTION:
XS GIS Cut Line= 3
      1365205.01      6842388.02       1365053.4      6842141.86
      1364554.99      6841537.98
#Sta/Elev= 30
  4710.9 2230.55  4776.6 2223.58  4834.6 2219.99  4898.8 2219.29  4913.8 2213.85
  4929.8 2205.12  4942.1 2201.85  4942.6 2201.35  4958.8 2201.85  4965.9 2204.01
  4971.8 2202.36  4987.2 2208.48    4993 2207.67  5008.4 2210.76  5199.9 2212.17
  5236.5 2214.33  5256.8  2219.1  5278.1 2222.93  5306.8 2222.78  5349.8 2220.94
  5356.3 2217.98  5384.9 2214.15  5412.5 2216.42  5434.4 2216.11  5456.6 2221.09
    5486 2222.56  5541.3 2223.94    5613 2229.15  5633.8  2228.5    5783 2237.67
#Mann= 7 ,-1 , 0
  4710.9     .07       0  4929.8     .16       0  4942.1     .07       0
  4958.8     .16       0  5256.8     .07       0  5412.5     .16       0
    5486     .07       0
Bank Sta=4942.1,4958.8
XS Rating Curve= 0 ,0
Exp/Cntr=0.3,0.1

Type RM Length L Ch R = 1 ,14508   ,497,497,497
BEGIN DESCRIPTION:
Long Branch 26.0
END DESCRIPTION:
XS GIS Cut Line= 3
        1365455.      6842338.01      1365410.89      6841940.15
      1364805.01      6841338.01
#Sta/Elev= 30
  4599.7 2238.63    4640 2235.47    4645 2233.02  4680.2 2222.85  4700.3 2214.95
  4720.4 2210.16  4762.5 2209.67  4830.4 2209.49  4871.4 2209.39    4917 2206.92
  4961.9 2206.82    4972    2205  4981.7  2199.8  4983.8 2198.88  4984.3 2198.38
  5000.5 2198.88  5005.7 2204.51  5019.8 2206.23  5090.6 2208.89  5097.6 2210.85
  5116.5 2211.44  5189.5 2217.14    5239 2218.78  5366.3 2218.04  5507.7 2219.49
  5606.7 2226.38    5628 2226.09  5656.2 2229.02  5769.4 2235.35  5854.2 2241.77
#Mann= 7 ,-1 , 0
  4599.7     .07       0  4762.5     .16       0  4830.4     .07       0
  4981.7     .16       0  4983.8     .07       0  5000.5     .16       0
  5116.5     .07       0
Bank Sta=4983.8,5000.5
XS Rating Curve= 0 ,0
Exp/Cntr=0.3,0.1

Type RM Length L Ch R = 1 ,14011   ,493,493,493
BEGIN DESCRIPTION:
Long Branch 25.0
END DESCRIPTION:
XS GIS Cut Line= 3
        1365955.      6842138.01       1365875.6      6841938.64
      1365405.03      6841338.03
#Sta/Elev= 30
  4785.4 2223.13  4817.7  2220.5  4824.5 2218.74  4854.2 2217.22  4871.5 2214.42
  4914.6 2212.38  4925.3 2210.59  4932.4    2205  4946.9 2200.49  4979.2 2202.81
  4986.3 2199.62  4989.3 2195.81  4989.8 2195.31    5006 2195.81  5014.5 2201.73
  5022.6 2203.45  5046.3 2203.59  5072.3 2201.66  5078.7 2203.47  5101.2 2202.43
  5175.7 2205.46  5370.7 2212.19  5420.4  2211.3  5492.7  2205.8    5528 2205.34
  5598.5 2209.39  5627.4 2213.65  5741.4 2225.06  5749.5 2228.01    5763    2229
#Mann= 5 ,-1 , 0
  4785.4     .07       0  4989.3     .07       0    5006     .07       0
  5046.3     .16       0  5175.7     .07       0
Bank Sta=4989.3,5006
XS Rating Curve= 0 ,0
Exp/Cntr=0.3,0.1

Type RM Length L Ch R = 1 ,13518   ,454,454,454
BEGIN DESCRIPTION:
Long Branch 24.0
END DESCRIPTION:
XS GIS Cut Line= 3
      1366105.01      6841738.01      1365854.52       6841482.8
      1365754.98      6841287.96
#Sta/Elev= 30
  4642.4 2213.52  4698.9 2213.55  4755.5 2212.05  4812.1 2207.34  4840.4 2206.08
  4854.5 2204.79  4875.8 2204.51  4911.1 2202.22  4974.8 2200.22  4981.8 2199.77
  4988.9 2197.05    4996 2193.16  4999.9 2193.73  5002.1 2192.97  5002.6 2192.47
  5018.4 2192.47  5018.9 2192.97  5027.1 2193.29  5032.7 2194.89  5049.3 2194.57
  5054.9    2197  5077.1 2200.73    5116 2200.85  5138.2 2201.98    5166 2207.38
  5182.6  2211.7  5188.2 2211.79  5204.8 2216.46  5210.4 2215.65  5218.8 2216.61
#Mann= 3 ,-1 , 0
  4642.4     .07       0  5002.1     .07       0  5018.9     .07       0
Bank Sta=5002.1,5018.9
XS Rating Curve= 0 ,0
Exp/Cntr=0.3,0.1

Type RM Length L Ch R = 1 ,13064   ,981,981,981
BEGIN DESCRIPTION:
Long Branch 23.0
END DESCRIPTION:
XS GIS Cut Line= 3
        1366105.      6841587.97      1366078.06      6841114.14
      1365905.04      6840988.03
#Sta/Elev= 30
  4525.4 2211.38  4605.5 2209.95  4645.6  2208.5  4705.7 2205.48  4725.7 2203.63
  4805.8 2198.81  4865.9  2199.2    4886 2198.44    4896 2199.07    4916 2198.29
  4968.4 2199.23  4976.1  2198.9  4986.1 2194.52  4987.1 2191.75  4987.6 2191.25
    5004 2191.75    5006 2193.19  5014.4 2195.86  5020.6 2196.37  5028.5  2200.1
    5050 2201.56  5064.7 2204.78    5078 2209.71  5085.5 2213.77  5091.7 2214.63
  5106.4 2216.17  5150.4 2218.26  5156.6 2217.82  5171.3 2219.29  5214.1 2220.79
#Mann= 3 ,-1 , 0
  4525.4     .07       0  4987.1     .07       0    5004     .07       0
Bank Sta=4987.1,5004
XS Rating Curve= 0 ,0
Exp/Cntr=0.3,0.1

Type RM Length L Ch R = 1 ,12083   ,496,496,496
BEGIN DESCRIPTION:
Long Branch 22.0
END DESCRIPTION:
XS GIS Cut Line= 3
        1366855.      6841487.98      1366841.96      6841252.04
      1366254.97      6840637.97
#Sta/Elev= 30
  4763.7 2214.22  4841.1 2211.32  4873.9 2210.33  4883.9 2210.94  4939.4 2208.66
    4954 2206.99    4964 2203.61    4974  2195.3    4984 2188.51  4985.5  2186.1
    4986  2185.6  5002.5  2186.1  5007.7 2191.72  5014.9 2193.73  5029.1 2194.26
  5079.9 2192.83  5128.1 2193.67  5148.2 2194.83  5177.5 2196.36  5198.9 2198.81
  5276.6 2204.09    5319  2205.8  5389.8 2205.78  5432.3 2204.89  5509.9 2205.14
  5651.5 2208.12  5708.1 2210.68    5715 2211.58  5736.4 2211.93  5849.5 2220.25
#Mann= 7 ,-1 , 0
  4763.7     .07       0  4841.1    .035       0  4939.4     .07       0
  4985.5     .07       0  5002.5     .07       0  5079.9     .16       0
  5148.2     .07       0
Bank Sta=4985.5,5002.5
XS Rating Curve= 0 ,0
Exp/Cntr=0.3,0.1

Type RM Length L Ch R = 1 ,11587   ,992,992,992
BEGIN DESCRIPTION:
Long Branch 21.0
END DESCRIPTION:
XS GIS Cut Line= 3
        1367255.      6841388.02      1367184.94      6840988.01
      1366204.99      6840287.99
#Sta/Elev= 30
  4593.9  2209.8  4715.7 2207.84  4847.7 2203.74  4878.2 2201.09  4898.5 2194.08
  4918.8 2190.64  5007.3 2191.32  5013.5  2190.4  5019.7 2184.82  5020.2 2184.32
  5036.7 2184.82  5036.8 2185.52    5129 2196.35  5221.2 2200.84  5330.5 2202.48
  5416.6 2201.27  5559.1 2202.04  5594.8 2201.28    5666 2202.04    5725 2204.16
  5737.3 2205.66  5752.1 2205.26  5909.4 2217.43  5946.2  2220.8  5953.6 2222.68
  5983.1 2224.66  5989.2 2226.02  6024.9 2228.78  6104.7 2237.55  6204.3 2245.53
#Mann= 3 ,-1 , 0
  4593.9     .07       0  5019.7     .07       0  5036.7     .07       0
Bank Sta=5019.7,5036.7
XS Rating Curve= 0 ,0
Exp/Cntr=0.3,0.1

Type RM Length L Ch R = 1 ,10595   ,498,498,498
BEGIN DESCRIPTION:
Long Branch 20.0
END DESCRIPTION:
XS GIS Cut Line= 3
      1367604.99      6841187.96      1367401.48        6840487.
      1366805.03      6839888.03
#Sta/Elev= 30
  4270.1 2204.44  4537.3 2198.85  4734.5  2197.7  4832.4 2195.29  4884.4 2197.09
  4932.4 2195.22  4957.3 2192.54  4977.6 2187.48  4988.5 2185.17    5000 2184.39
  5002.4 2179.75  5002.9 2179.25  5019.5 2179.75  5032.2 2184.86  5039.2 2186.28
  5088.7 2185.83  5102.9 2186.78  5138.2 2185.56    5206 2187.33  5230.1 2188.73
  5258.4 2193.01  5265.5 2192.39  5272.6 2193.83  5279.7 2192.89  5286.7 2194.11
  5293.8 2193.11  5307.9 2193.59  5654.4 2209.68  5795.8 2222.31  5845.3 2225.41
#Mann= 6 ,-1 , 0
  4270.1     .07       0  4734.5     .16       0  4977.6     .12       0
  5002.4     .07       0  5019.5     .12       0    5206     .07       0
Bank Sta=5002.4,5019.5
XS Rating Curve= 0 ,0
Exp/Cntr=0.3,0.1

Type RM Length L Ch R = 1 ,10097   ,497,497,497
BEGIN DESCRIPTION:
Long Branch 19.0
END DESCRIPTION:
XS GIS Cut Line= 3
      1367854.99      6841237.97      1367357.25      6840131.58
      1367455.02      6839937.96
#Sta/Elev= 30
  3786.8 2206.74    3876 2205.61  3907.4 2203.52  3916.9 2204.21  3968.6 2202.11
  3984.1 2203.08  4234.3 2197.66  4460.9 2196.08  4557.2 2194.96  4603.5 2192.87
    4637 2189.69    4673 2186.57  4807.3 2185.41    4834 2185.34  5007.8 2183.23
  5024.5  2180.7  5030.1  2181.5  5037.6 2180.08  5038.2 2177.92  5038.7 2177.42
  5055.4 2177.92    5060 2178.17  5069.1 2181.24  5074.7 2180.46  5091.4 2186.49
  5119.3 2193.56  5141.6 2195.76  5175.6 2201.24  5194.4 2203.05  5216.9 2203.06
#Mann= 8 ,-1 , 0
  3786.8     .07       0  4460.9     .16       0    4637     .12       0
  4807.3     .16       0    4834     .12       0  5038.2     .07       0
  5055.4     .12       0  5175.6     .07       0
Bank Sta=5038.2,5055.4
XS Rating Curve= 0 ,0
Exp/Cntr=0.3,0.1

Type RM Length L Ch R = 1 ,9600    ,496,496,496
BEGIN DESCRIPTION:
Long Branch 18.0
END DESCRIPTION:
XS GIS Cut Line= 3
        1367855.      6840987.98      1367774.98      6840288.04
        1367705.      6839737.97
#Sta/Elev= 30
  4295.5 2201.39    4376  2199.6  4406.2 2197.94  4436.4 2197.87  4466.6 2195.19
  4513.7 2193.85    4527 2194.43  4587.4 2193.24  4748.4 2194.09  4775.4  2192.9
  4781.7 2193.82  4808.8 2192.91  4848.1 2189.42  4889.3 2184.38  4939.6 2182.97
  4949.7 2181.98  4960.3 2180.24  4961.2 2176.15  4961.7 2175.65  4978.4 2176.15
  4997.5 2181.59  5030.3 2183.09  5050.4 2188.34  5060.5 2189.96  5181.7 2194.48
  5357.2 2200.55  5362.9 2201.79  5413.3 2205.17  5504.1 2214.91  5554.5 2222.49
#Mann= 6 ,-1 , 0
  4295.5     .07       0  4775.4     .16       0  4848.1     .12       0
  4961.2     .07       0  4978.4     .12       0  5181.7     .07       0
Bank Sta=4961.2,4978.4
XS Rating Curve= 0 ,0
Exp/Cntr=0.3,0.1

Type RM Length L Ch R = 1 ,9104    ,497,497,497
BEGIN DESCRIPTION:
Long Branch 17.0
END DESCRIPTION:
XS GIS Cut Line= 3
       1367945.6      6841004.55      1368239.28      6840288.97
      1368104.99      6839787.96
#Sta/Elev= 30
  4226.5  2202.1  4393.2 2192.55  4601.1 2190.93    4684 2189.17  4744.9 2186.28
  4761.3 2184.08  4790.7 2182.61  4806.5 2179.61  4814.7  2181.4  4873.5 2177.82
  4921.1  2179.4  4957.8 2181.11  4968.6 2179.49  4971.6 2172.75  4972.1 2172.25
  4988.8 2172.75  4997.8 2176.03  5003.1 2176.03  5011.4 2179.07  5021.7 2180.75
  5036.5 2180.32  5071.4 2184.64  5076.6 2183.62  5125.2 2188.05  5306.3 2191.28
  5394.4 2196.45  5404.8 2195.96  5426.4 2199.31  5461.2 2207.32  5518.7  2211.5
#Mann= 5 ,-1 , 0
  4226.5     .07       0  4744.9     .16       0  4921.1     .07       0
  4971.6     .07       0  4988.8     .07       0
Bank Sta=4971.6,4988.8
XS Rating Curve= 0 ,0
Exp/Cntr=0.3,0.1

Type RM Length L Ch R = 1 ,8607    ,479,479,479
BEGIN DESCRIPTION:
Long Branch 16.0
END DESCRIPTION:
XS GIS Cut Line= 3
      1368554.99      6840937.96      1368454.77      6840222.85
      1368305.01      6839688.02
#Sta/Elev= 30
  4277.9 2201.18  4429.3 2191.64  4461.3 2188.04  4479.8 2181.93  4510.1 2175.45
  4520.2 2178.86  4590.9 2178.31  4621.2 2183.57  4681.8 2186.23  4784.5 2182.14
  4974.6  2176.4  4984.7 2174.51  4986.2 2171.05  4986.7 2170.55  5003.4 2171.05
  5005.1 2174.81  5009.2 2174.71    5014 2174.59  5019.1 2177.77  5046.6 2177.43
  5077.7 2180.93  5087.4  2179.7  5092.6 2183.29    5140  2186.1  5244.6 2187.92
  5264.7 2184.92  5420.4 2196.23  5430.8  2199.6  5482.7 2207.38  5555.4 2213.03
#Mann= 5 ,-1 , 0
  4277.9     .07       0  4784.5     .16       0  4986.2     .07       0
  5003.4     .16       0  5009.2     .07       0
Bank Sta=4986.2,5003.4
XS Rating Curve= 0 ,0
Exp/Cntr=0.3,0.1

Type RM Length L Ch R = 1 ,8128    ,784,784,784
BEGIN DESCRIPTION:
Long Branch 15.0
END DESCRIPTION:
XS GIS Cut Line= 3
        1368655.      6840938.03      1368720.33      6840337.38
      1368604.99      6839737.97
#Sta/Elev= 30
  4395.8 2202.67  4436.1  2201.4  4466.2 2197.02  4526.6 2192.56  4687.5 2185.07
  4747.9 2183.82  4778.1  2181.2  4807.6 2182.18  4818.3 2184.41  4838.4 2184.35
  4858.5 2177.81  4904.1 2177.63    4929 2180.96  4952.6 2179.97  4959.1 2179.48
  4980.3 2171.47  4980.8 2170.97  4998.3 2171.47  4998.5 2175.25  5009.5 2176.13
  5040.1 2174.92  5071.4 2176.36  5121.6 2178.96    5203 2179.59  5274.3 2184.33
  5423.6 2185.93  5508.5 2188.95  5532.5 2190.74  5584.4 2200.39  5610.4 2209.96
#Mann= 5 ,-1 , 0
  4395.8     .07       0  4952.6     .16       0  4980.3     .07       0
  4998.3     .16       0  5071.4     .07       0
Bank Sta=4980.3,4998.3
XS Rating Curve= 0 ,0
Exp/Cntr=0.3,0.1

Type RM Length L Ch R = 1 ,7344    ,127,127,127
BEGIN DESCRIPTION:
Long Branch 14.0
END DESCRIPTION:
XS GIS Cut Line= 3
      1368948.62      6840916.67      1369104.73      6840413.11
      1369173.33      6839724.62
#Sta/Elev= 30
  4472.8 2198.79  4574.8 2194.94  4645.2 2189.03  4650.5 2189.99  4742.8 2183.49
  4916.4 2175.13  4932.1  2177.1  4942.5 2176.58  4973.9  2171.3  4977.8 2168.73
  4978.3 2168.23  4995.9 2168.73    5000 2170.72  5025.2 2173.11  5045.3 2173.19
  5051.8 2171.46  5056.8 2173.16  5145.8 2175.28  5152.4 2175.86  5157.5 2178.51
  5206.1 2182.63    5387 2181.61  5517.7 2184.18  5555.2 2187.86  5560.2 2186.82
    5588  2190.2  5638.3 2192.65  5660.9 2195.03  5668.4    2197  5691.9 2197.29
#Mann= 4 ,-1 , 0
  4472.8    .035       0  4742.8     .07       0  4977.8     .07       0
  4995.9     .07       0
Bank Sta=4977.8,4995.9
XS Rating Curve= 0 ,0
Exp/Cntr=0.3,0.1

Type RM Length L Ch R = 1 ,7217    ,532,532,532
BEGIN DESCRIPTION:
Long Branch 13.0
END DESCRIPTION:
XS GIS Cut Line= 3
        1369105.        6840888.      1369178.27      6840511.36
        1369255.      6839588.04
#Sta/Elev= 30
  4616.3  2194.1  4728.4 2190.14  4750.5 2186.73  4809.9 2182.17  4860.8 2176.86
  4905.5 2174.03  4957.1 2172.62    4974 2169.84  4974.5 2169.34  4992.1 2169.84
  5145.3 2180.61    5184 2181.51  5234.2 2180.52  5265.9 2181.93  5284.3 2181.23
  5324.5 2182.15    5450 2181.74  5463.3 2181.84  5575.3 2181.97  5655.6 2184.51
  5735.9 2189.69  5743.2 2191.25  5748.2 2190.36  5776.3 2194.56  5797.5 2197.52
  5816.2 2200.03  5856.3 2202.67  5868.8 2202.48  5896.4 2204.91  5926.5 2205.99
#Mann= 7 ,-1 , 0
  4616.3     .07       0    4974     .07       0  4992.1     .07       0
    5450     .16       0  5463.3     .07       0  5776.3    .035       0
  5797.5     .07       0
Bank Sta=4974,4992.1
XS Rating Curve= 0 ,0
Exp/Cntr=0.3,0.1

Type RM Length L Ch R = 1 ,6685    ,498,498,498
BEGIN DESCRIPTION:
Long Branch 12.0
END DESCRIPTION:
XS GIS Cut Line= 3
      1369805.02      6840638.01      1369515.49      6840489.49
      1369305.01      6839588.03
#Sta/Elev= 30
  4674.6 2194.68  4675.7 2194.68  4688.5  2193.1  4727.3 2179.79  4749.5  2175.7
  4771.7 2175.58  4777.3 2178.21  4793.9 2178.87  4799.5 2182.54  4816.1  2183.8
  4821.7 2188.01  4860.5 2187.92  4866.1 2183.85  4876.9 2185.02  4888.3 2183.33
  4910.6 2175.39  4952.2    2170  4978.9 2165.21  4979.4 2164.71    4997 2165.21
  4997.5 2172.44  5115.9  2178.6  5510.3 2179.57  5596.8 2181.15    5679 2183.95
  5747.9 2190.12  5762.7 2191.98  5811.7  2197.1  5843.6 2196.95  5925.7 2205.72
#Mann= 9 ,-1 , 0
  4674.6     .07       0  4675.7     .16       0  4952.2     .07       0
  4978.9     .07       0    4997     .07       0  5510.3     .16       0
  5596.8     .07       0  5747.9    .035       0  5762.7     .07       0
Bank Sta=4978.9,4997
XS Rating Curve= 0 ,0
Exp/Cntr=0.3,0.1

Type RM Length L Ch R = 1 ,6187    ,320,320,320
BEGIN DESCRIPTION:
Long Branch 11.0
END DESCRIPTION:
XS GIS Cut Line= 3
        1369855.      6840588.01      1369928.36      6840264.73
        1369805.      6839687.98
#Sta/Elev= 30
  4668.5 2194.82  4699.3 2193.07  4709.5 2191.15  4735.7 2183.83  4750.5 2182.29
  4760.8 2177.59  4778.8 2171.93  4791.6  2170.6  4832.6 2168.34  4918.4 2170.55
  4945.4 2165.27  4961.5 2164.78  4966.6 2167.44    5000 2166.75  5006.9 2165.12
  5008.1  2163.3  5008.6  2162.8  5026.2  2163.3  5027.3 2166.51  5036.2 2170.17
  5041.3 2168.84  5109.1 2175.21  5354.6  2175.4  5455.5 2177.27  5473.8  2178.2
  5515.6 2179.94  5548.9 2183.28  5559.1 2185.63    5565 2189.07  5589.8 2193.01
#Mann= 5 ,-1 , 0
  4668.5     .07       0  5008.1     .07       0  5026.2     .07       0
  5455.5     .16       0  5473.8     .07       0
Bank Sta=5008.1,5026.2
XS Rating Curve= 0 ,0
Exp/Cntr=0.3,0.1

Type RM Length L Ch R = 1 ,5867    ,158,158,158
BEGIN DESCRIPTION:
Long Branch 10.1
END DESCRIPTION:
XS GIS Cut Line= 3
      1370069.14      6840670.85      1370171.66      6840104.25
      1370117.99      6839490.99
#Sta/Elev= 30
  4424.2 2185.08  4457.6  2184.3  4569.4 2178.48  4654.7 2177.46  4772.6  2177.4
  4864.1 2172.87  4873.7 2173.88  4878.8 2172.02  4894.6 2170.04  4904.7 2169.84
  4937.4 2165.92  4955.5 2165.95  5006.1 2162.64  5006.6 2162.14  5024.3 2162.64
  5046.4 2164.16  5086.6 2170.12  5137.8 2173.62    5187 2173.73  5257.2 2175.78
  5312.5 2174.23  5377.7 2174.23  5407.8 2175.45  5437.9 2177.66  5463.3  2181.6
  5467.2  2182.6  5475.5 2186.49  5480.5 2185.84  5488.1 2190.09  5615.6 2191.41
#Mann= 6 ,-1 , 0
  4424.2     .07       0  5006.1     .07       0  5024.3     .07       0
  5312.5     .16       0  5463.3     .07       0  5467.2    .035       0
Bank Sta=5006.1,5024.3
XS Rating Curve= 0 ,0
Exp/Cntr=0.3,0.1

Type RM Length L Ch R = 1 ,5709    ,333,333,333
BEGIN DESCRIPTION:
Long Branch 10.0
END DESCRIPTION:
XS GIS Cut Line= 3
      1370141.73      6840783.79      1370296.49      6840185.38
      1370244.29      6839497.06
#Sta/Elev= 30
  4381.9 2184.95  4430.3 2184.64  4576.8 2181.09  4612.3 2179.33  4617.5 2179.89
  4652.9 2177.63  4658.1 2178.39  4693.5 2176.86  4883.7 2176.59  4932.1 2171.93
  4966.3 2170.07  4972.8 2168.73  4977.9 2169.94    5000  2168.3  5047.5 2163.08
  5067.6 2163.11  5068.5 2161.99    5069 2161.49  5086.7 2161.99  5117.7 2163.58
  5187.9 2170.69  5403.9 2174.22  5408.7 2174.27  5483.1 2175.25    5549  2179.4
  5639.2 2186.93  5648.4 2189.29  5659.3 2190.74  5669.3 2193.47  5690.3 2193.66
#Mann= 7 ,-1 , 0
  4381.9    .035       0  4430.3     .07       0  5068.5     .07       0
  5086.7     .07       0  5403.9     .16       0  5408.7     .07       0
  5648.4    .035       0
Bank Sta=5068.5,5086.7
XS Rating Curve= 0 ,0
Exp/Cntr=0.3,0.1

Type RM Length L Ch R = 1 ,5376    ,166,166,166
BEGIN DESCRIPTION:
Long Branch 9.1
END DESCRIPTION:
XS GIS Cut Line= 3
      1370561.39      6840921.47      1370525.34      6839968.06
      1370498.43      6839578.98
#Sta/Elev= 30
  4045.9 2177.55  4169.5 2176.38  4229.5 2177.04  4339.6 2174.56  4359.6 2175.46
  4399.6  2173.9  4429.6 2174.76  4459.7 2172.82  4599.8 2170.44  4613.4 2171.78
  4659.8 2170.46  4819.9 2169.89  4880.8 2172.32    4960 2168.03    4980 2165.93
  5002.5 2162.95    5011 2156.94  5011.5 2156.44  5029.2 2156.94  5030.1 2158.87
  5050.2 2163.13  5100.3 2164.78  5200.5 2171.82  5310.8 2176.56  5340.9 2181.66
  5350.9 2186.14  5360.9 2184.76  5371.6 2186.31    5388 2179.43    5390 2179.43
#Mann= 3 ,-1 , 0
  4045.9     .07       0    5011     .07       0  5029.2     .07       0
Bank Sta=5011,5029.2
XS Rating Curve= 0 ,0
Exp/Cntr=0.3,0.1

Type RM Length L Ch R = 1 ,5210    ,456,456,456
BEGIN DESCRIPTION:
Long Branch 9.0
END DESCRIPTION:
XS GIS Cut Line= 3
      1370673.55      6840950.64       1370639.6      6839887.28
      1370617.11      6839323.93
#Sta/Elev= 30
  3936.1  2178.7  4018.8 2177.41  4118.8 2173.28  4198.9 2172.94    4529 2166.79
  4639.1 2166.16  4669.1 2167.04  4674.1 2168.52  4779.2 2167.16  4829.2 2165.14
  4969.3 2164.11  4979.3 2163.74  4985.8 2162.14    4988 2155.25  4988.5 2154.75
  5006.2 2155.25  5019.3 2160.96  5029.3 2167.35  5039.3 2169.15  5119.4 2174.26
  5149.4 2177.78  5179.4 2178.67  5229.5 2176.86  5329.2 2176.93  5330.6 2176.97
  5409.6 2178.51  5519.7 2177.97  5539.7 2179.04  5559.2 2183.53  5563.8 2183.53
#Mann= 5 ,-1 , 0
  3936.1     .07       0    4988     .07       0  5006.2     .07       0
  5329.2    .035       0  5330.6     .07       0
Bank Sta=4988,5006.2
XS Rating Curve= 0 ,0
Exp/Cntr=0.3,0.1

Type RM Length L Ch R = 1 ,4754    ,497,497,497
BEGIN DESCRIPTION:
Long Branch 8.0
END DESCRIPTION:
XS GIS Cut Line= 3
      1370705.01      6840687.98      1370980.14      6840038.56
        1371005.      6839737.98
#Sta/Elev= 30
  4294.7 2173.77  4303.8 2173.05    4349 2173.34    4362 2172.19  4409.4 2171.63
    4425 2172.37  4446.7 2171.04  4522.7 2170.12  4849.9 2167.94  4868.2 2169.05
  4891.8 2168.21  4913.9 2168.56  4950.1 2168.29  4973.7 2166.98  4979.2 2167.88
  4989.7 2163.99  4997.4 2160.14  5001.5 2152.33    5002 2151.83  5019.7 2152.33
  5020.6 2155.24  5030.7 2157.65  5040.7 2158.48  5050.7 2162.06  5090.9 2163.04
  5145.8 2166.04  5238.6 2170.27  5261.4 2169.99  5291.5 2183.25  5301.6 2182.33
#Mann= 5 ,-1 , 0
  4294.7     .07       0  4913.9     .16       0  5001.5     .07       0
  5019.7     .16       0  5145.8     .07       0
Bank Sta=5001.5,5019.7
XS Rating Curve= 0 ,0
Exp/Cntr=0.3,0.1

Type RM Length L Ch R = 1 ,4257    ,497,497,497
BEGIN DESCRIPTION:
Long Branch 7.0
END DESCRIPTION:
XS GIS Cut Line= 3
      1370750.99      6840848.75      1371313.42      6840193.94
      1371288.65       6839727.1
#Sta/Elev= 30
  4136.8 2174.57  4282.5  2172.7  4360.4 2170.49  4452.6 2170.01  4473.4 2168.98
  4686.3 2167.24  4707.2 2165.85    4807 2164.43  4845.7 2161.47    4863 2160.65
  4913.5 2161.99  4948.6 2160.47  4955.2 2156.28  4969.5 2155.06  4977.1 2155.89
  4991.4 2155.12  4997.4 2153.41  5016.8 2151.44  5017.3 2150.94  5035.1 2151.44
    5046 2155.06  5062.8 2158.71  5067.8 2155.68    5076 2158.95  5086.1 2158.26
  5106.1 2159.23  5146.1 2163.51  5197.7 2166.07  5246.3  2167.6  5467.5 2166.21
#Mann= 5 ,-1 , 0
  4136.8     .07       0  4845.7     .16       0  5016.8     .07       0
  5035.1     .16       0  5197.7     .07       0
Bank Sta=5016.8,5035.1
XS Rating Curve= 0 ,0
Exp/Cntr=0.3,0.1

Type RM Length L Ch R = 1 ,3760    ,499,499,499
BEGIN DESCRIPTION:
Long Branch 6.0
END DESCRIPTION:
XS GIS Cut Line= 3
      1371354.98      6840788.04      1371652.91      6840191.16
       1371591.9      6839715.56
#Sta/Elev= 30
  4332.9  2175.2  4346.9 2172.37  4430.8 2170.36  4511.8 2166.37  4712.9 2164.01
  4757.7 2162.89  4766.4  2161.9  4794.4 2162.73  4833.5 2158.79  4839.1 2159.75
  4855.9 2158.85  4861.5 2160.63  4878.3 2155.76  4883.9 2155.87  4891.8 2153.47
  4896.1 2153.31  4958.8 2153.64  4967.8 2152.44    4972  2148.7  4972.5  2148.2
  4990.3  2148.7  4995.7 2148.98    4999 2154.93  5004.1 2154.93  5033.4 2160.93
  5055.9 2163.11  5134.3 2164.78    5225  2164.6  5295.6 2165.97  5479.5 2163.43
#Mann= 5 ,-1 , 0
  4332.9     .07       0  4896.1     .16       0    4972     .07       0
  4990.3     .16       0  5055.9     .07       0
Bank Sta=4972,4990.3
XS Rating Curve= 0 ,0
Exp/Cntr=0.3,0.1

Type RM Length L Ch R = 1 ,3261    ,500,500,500
BEGIN DESCRIPTION:
Long Branch 5.0
END DESCRIPTION:
XS GIS Cut Line= 3
        1371805.      6840987.99      1371858.74      6840586.48
      1372036.54      6840408.45
#Sta/Elev= 30
  4594.9 2181.17  4625.2 2175.62  4631.4 2174.15  4636.4 2171.58  4655.4 2169.99
  4675.6 2170.81  4685.7 2169.53  4695.8  2165.7  4704.4 2164.04  4726.1 2161.15
  4826.9 2159.41  4897.6 2161.58  4927.8 2159.53  4938.5 2154.96  4958.1 2150.18
  4969.1 2145.63  4969.6 2145.13  4987.4 2145.63    5000 2147.83  5003.3 2154.66
  5010.4 2154.06  5017.5 2155.58  5038.7  2154.9  5045.8 2155.92  5052.8 2152.94
  5059.9    2155    5067 2154.87  5109.4 2160.09  5151.8 2162.03  5251.6 2160.93
#Mann= 3 ,-1 , 0
  4594.9     .07       0  4969.1     .07       0  4987.4     .07       0
Bank Sta=4969.1,4987.4
XS Rating Curve= 0 ,0
Exp/Cntr=0.3,0.1

Type RM Length L Ch R = 1 ,2761    ,498,498,498
BEGIN DESCRIPTION:
Long Branch 4.0
END DESCRIPTION:
XS GIS Cut Line= 3
      1371912.18      6841057.65      1372191.22      6840824.85
      1372225.92      6840475.97
#Sta/Elev= 30
  4636.6 2175.05  4645.3 2175.91  4653.1 2173.37  4666.3 2172.81  4680.5 2167.68
  4702.6 2163.78  4744.5 2160.07  4766.4 2160.01  4787.2 2157.53    4795 2157.95
  4801.5 2156.05  4836.7  2154.3  4844.5 2151.94  4873.1 2154.65  4908.2 2152.71
  4922.6 2153.69  4936.9 2152.32  4965.5 2152.62    4972 2151.42  4977.2 2142.62
  4977.7 2142.12  4995.5 2142.62  4999.2 2151.06  5016.9 2152.82  5071.9 2154.48
  5085.5 2154.69  5090.5 2157.25  5147.6 2159.19  5232.1 2158.16  5350.6 2159.45
#Mann= 5 ,-1 , 0
  4636.6     .07       0  4977.2     .07       0  4995.5     .07       0
  5071.9     .16       0  5232.1     .07       0
Bank Sta=4977.2,4995.5
XS Rating Curve= 0 ,0
Exp/Cntr=0.3,0.1

Type RM Length L Ch R = 1 ,2263    ,498,498,498
BEGIN DESCRIPTION:
Long Branch 3.0
END DESCRIPTION:
XS GIS Cut Line= 3
      1372155.01        6841288.      1372391.93      6841224.03
      1372387.59      6840588.95
#Sta/Elev= 30
  4754.6 2182.99  4757.2 2182.99  4764.9 2178.75  4771.9 2176.67  4777.1 2178.06
    4796 2177.21  4811.8 2178.28    4817 2177.64  4837.5 2169.27  4846.6 2167.81
  4858.2 2163.61  4886.5 2161.63  4891.6 2158.31  4899.6 2156.51  4931.5 2155.57
    4941 2152.91  4982.5 2149.24  4992.8 2147.36  4996.8 2141.59  4997.3 2141.09
  5015.2 2141.59    5016 2148.07    5026 2150.35    5056 2152.61    5096 2153.62
    5116 2155.17  5164.9 2155.13    5332 2155.55  5575.4 2156.91  5635.1 2157.31
#Mann= 6 ,-1 , 0
  4754.6     .07       0  4996.8     .07       0  5015.2     .07       0
  5164.9     .07       0    5332     .16       0  5575.4     .07       0
Bank Sta=4996.8,5015.2
XS Rating Curve= 0 ,0
Exp/Cntr=0.3,0.1

Type RM Length L Ch R = 1 ,1765    ,492,492,492
BEGIN DESCRIPTION:
Long Branch 2.0
END DESCRIPTION:
XS GIS Cut Line= 3
      1372554.99      6841588.01      1372855.03      6841338.08
      1372869.58      6840814.38
#Sta/Elev= 30
  4609.5 2181.66  4612.8 2181.66  4616.7 2177.95    4631 2173.49  4651.8 2163.87
    4674 2158.45  4709.1 2154.77  4822.3 2152.48  4830.2 2149.95  4843.8 2149.05
    4851 2150.99  4857.5 2149.09  4865.3 2151.57  4879.6 2152.23  4888.2 2150.97
  4964.2 2146.35  4972.1 2147.84  4978.6 2141.36  4986.4  2140.9  4987.5  2139.2
    4988  2138.7  5005.9  2139.2  5010.1 2144.29  5020.1  2147.8  5100.1 2150.38
    5151 2149.74  5156.8  2150.1  5190.1  2151.6  5395.5 2152.96  5523.9 2153.64
#Mann= 7 ,-1 , 0
  4609.5     .07       0  4888.2     .16       0  4987.5     .07       0
  5005.9     .16       0    5151     .07       0  5156.8     .16       0
  5395.5     .07       0
Bank Sta=4987.5,5005.9
XS Rating Curve= 0 ,0
Exp/Cntr=0.3,0.1

Type RM Length L Ch R = 1 ,1273    ,427,427,427
BEGIN DESCRIPTION:
Long Branch 1.0
END DESCRIPTION:
XS GIS Cut Line= 3
      1372955.03      6841687.97      1373315.19      6841337.55
      1373280.62      6841193.95
#Sta/Elev= 30
  4497.5 2158.61  4511.5 2156.44  4518.7 2156.27  4525.7 2152.21  4539.8 2151.32
    4646 2150.01  4723.7 2150.96  4822.7 2147.33    4851 2147.93  4872.3  2146.5
  4879.3 2147.29  4907.6  2146.1  4928.9 2146.75  4935.9 2148.61  4943.1 2147.85
    4950 2148.89  4957.2 2146.52  4971.4 2146.66  4978.3  2144.8  4983.3 2135.54
  4983.8 2135.04  5001.7 2135.54  5009.8 2141.75  5018.6  2146.4  5023.7 2146.26
  5030.4 2149.76  5040.7 2152.77  5060.5 2154.49  5107.6 2155.17  5147.7 2154.62
#Mann= 3 ,-1 , 0
  4497.5     .07       0  4983.3     .07       0  5001.7     .07       0
Bank Sta=4983.3,5001.7
XS Rating Curve= 0 ,0
Exp/Cntr=0.3,0.1
