HEC-RAS study Stink Creek.prj: Stink Creek Base Level Engineering

--- Stink Creek.g01 (geometry) --- (continued)

Type RM Length L Ch R = 1 ,37278   ,85,85,85
BEGIN DESCRIPTION:
Stink Creek 69.0
END DESCRIPTION:
XS GIS Cut Line= 6
      1441854.19      6856583.43      1441866.22      6857072.66
      1441501.32      6857098.87      1441178.76      6856846.86
      1441114.96      6856846.86      1440932.21      6856721.84
#Sta/Elev= 30
  4238.6 2054.75  4359.4  2053.7  4457.4 2053.31  4603.4 2052.34  4769.3  2050.8
  4779.3 2046.05  4799.3  2039.4  4909.5 2039.46  4969.6 2041.72  5019.8 2041.57
  5036.2 2042.97  5041.2 2046.23  5122.8 2047.13  5188.6 2047.12  5194.2  2039.4
  5194.7  2038.9  5207.1  2039.4  5210.5 2047.19    5219 2047.29  5295.4 2047.11
  5354.4  2049.7  5440.4 2047.63  5469.3 2047.83  5500.7  2049.7  5529.8 2049.01
  5576.3 2050.66  5597.3 2048.96  5618.3 2050.92    5669 2050.89  5791.3  2054.2
#Mann= 10 ,-1 , 0
  4238.6     .07       0  4359.4     .16       0  4457.4    .033       0
  4603.4     .16       0  5194.2     .07       0  5207.1     .16       0
    5219     .07       0  5354.4     .16       0  5440.4     .07       0
  5469.3     .16       0
Bank Sta=5194.2,5207.1
XS Rating Curve= 0 ,0
Exp/Cntr=0.3,0.1

Type RM Length L Ch R = 1 ,37193   ,193,193,193
BEGIN DESCRIPTION:
Stink Creek 4141
END DESCRIPTION:
XS GIS Cut Line= 6
      1440902.17      6856752.17      1441114.01       6856863.3
      1441179.98       6856863.3       1441383.1      6857047.33
      1441537.62      6857132.39      1441866.09      6857171.87
#Sta/Elev= 30
  4127.4 2054.06  4132.7 2053.04  4193.2 2053.83  4259.4 2050.08  4266.1 2050.91
  4319.9 2049.35    4364 2050.49    4458  2047.7  4467.7 2047.57  4510.1 2047.63
  4545.8 2049.36  4598.6 2048.51  4609.4 2048.96  4630.3 2047.08  4702.9 2047.16
  4840.7 2046.34  4841.2 2045.84  4853.7 2046.34  4883.1 2049.98  4891.8  2052.7
    4969 2050.56    4974 2052.22  4981.1 2052.31  5051.2 2050.43  5056.2 2052.14
  5132.2 2049.88  5138.4 2049.92  5143.4 2051.81  5162.4 2051.91  5213.9 2049.24
#Mann= 7 ,-1 , 0
  4127.4     .16       0    4458     .07       0  4467.7     .16       0
  4598.6     .07       0  4702.9     .16       0  4840.7     .07       0
  4853.7     .16       0
Bank Sta=4840.7,4853.7
XS Rating Curve= 0 ,0
Exp/Cntr=0.3,0.1

Type RM Length L Ch R = 1 ,37000   ,547,547,547
BEGIN DESCRIPTION:
Stink Creek 68.0
END DESCRIPTION:
XS GIS Cut Line= 3
        1440755.        6857188.      1441604.93      6857306.85
      1441870.48      6857184.69
#Sta/Elev= 30
  4141.8 2059.19  4212.5  2058.6  4293.3 2055.67  4313.5 2051.48  4320.4 2048.51
  4343.7 2042.24    4374 2039.56  4454.8    2039    4545 2041.34    4677  2043.8
  4707.2 2045.45  4737.5 2044.87  4754.1 2042.74  4759.2 2043.26  4798.1 2040.96
  4909.2 2044.56  4949.6 2040.85  4973.5 2039.64    4990 2040.14  4997.5    2036
    5000    2036  5000.9 2033.23  5001.4 2032.73  5013.9 2033.23  5030.4 2037.27
  5150.7 2039.07  5231.2 2044.34  5271.1 2047.93  5276.6 2049.55  5292.3 2048.07
#Mann= 4 ,-1 , 0
  4141.8     .07       0    4545     .16       0  5000.9     .07       0
  5013.9     .16       0
Bank Sta=5000.9,5013.9
XS Rating Curve= 0 ,0
Exp/Cntr=0.3,0.1

Type RM Length L Ch R = 1 ,36453   ,453,453,453
BEGIN DESCRIPTION:
Stink Creek 67.1
END DESCRIPTION:
XS GIS Cut Line= 3
      1440927.48      6857448.35      1441224.91      6857617.97
       1441601.8      6857593.31
#Sta/Elev= 30
  4657.6 2052.34  4663.5 2052.52    4707 2050.87  4712.7 2049.93  4728.6 2049.41
  4744.4 2047.33  4750.2 2047.99  4756.3 2047.46    4766 2046.43  4809.2 2046.34
  4868.3 2043.94  4933.1 2042.44  4942.5 2041.73  4948.9 2040.15  4954.7 2040.82
  4964.8  2038.4  4970.6  2038.1  4990.6 2032.59  4991.1 2032.09  5003.7 2032.59
  5020.1 2032.98  5030.2  2035.1  5050.2 2035.54  5130.4 2034.77  5170.5 2036.76
  5185.6 2038.38  5270.7 2040.53  5300.7 2042.04  5330.8 2045.21  5377.7 2047.25
#Mann= 6 ,-1 , 0
  4657.6     .07       0  4663.5     .16       0  4756.3     .07       0
  4990.6     .07       0  5003.7     .07       0  5185.6     .16       0
Bank Sta=4990.6,5003.7
XS Rating Curve= 0 ,0
Exp/Cntr=0.3,0.1

Type RM Length L Ch R = 1 ,36000   ,286,286,286
BEGIN DESCRIPTION:
Stink Creek 67.0
END DESCRIPTION:
XS GIS Cut Line= 3
        1440855.        6857888.      1441355.28      6857914.79
      1441576.74      6857634.78
#Sta/Elev= 30
    4499 2051.63  4565.7 2047.86  4591.6 2046.39  4729.3 2040.78  4769.4 2036.65
  4823.3 2036.96  4849.5 2036.65  4869.5 2039.34  4919.6 2034.47  4989.7    2033
  5004.7 2028.81  5005.2 2028.31    5018 2028.81  5025.8 2034.09  5040.2 2036.23
    5061 2037.23  5112.2 2037.44  5133.2  2037.4  5147.6 2038.49    5154 2040.44
  5161.7 2040.47  5168.4 2038.96  5174.8 2040.47  5182.9 2039.41  5189.2 2041.13
  5197.3 2040.73  5218.1 2042.55    5247 2042.38  5282.2 2045.76    5357 2046.68
#Mann= 7 ,-1 , 0
    4499     .16       0  4565.7     .07       0  4591.6     .16       0
  4823.3     .07       0  5004.7     .07       0    5018     .07       0
  5112.2     .16       0
Bank Sta=5004.7,5018
XS Rating Curve= 0 ,0
Exp/Cntr=0.3,0.1

Type RM Length L Ch R = 1 ,35714   ,489,489,489
BEGIN DESCRIPTION:
Stink Creek 66.2
END DESCRIPTION:
XS GIS Cut Line= 3
      1441187.79      6858314.24      1441365.32      6858198.18
       1441634.6      6857694.44
#Sta/Elev= 30
  4787.9 2041.99  4820.4 2042.21  4832.5 2041.39  4941.2 2042.28  4956.2 2042.02
  4967.6 2040.91  4992.4 2037.03  4996.8 2034.32  5002.9 2034.32  5013.6 2028.57
  5016.2 2028.31  5016.7 2027.81    5029 2027.81  5029.5 2028.31  5029.8 2029.42
  5035.5 2032.51  5045.6 2032.85  5152.8 2032.39  5183.5 2032.94  5205.4 2035.19
  5233.1 2035.54  5256.9 2035.41  5281.8 2035.82  5309.5 2037.74  5375.3 2040.73
  5413.5 2040.46  5515.3 2044.22  5555.8 2045.63  5561.1 2045.21  5571.2 2045.71
#Mann= 10 ,-1 , 0
  4787.9     .07       0  4941.2     .16       0  4967.6     .07       0
  5016.2     .07       0  5029.5     .07       0  5152.8     .16       0
  5233.1     .07       0  5256.9     .16       0  5515.3     .07       0
  5561.1     .16       0
Bank Sta=5016.2,5029.5
XS Rating Curve= 0 ,0
Exp/Cntr=0.3,0.1

Type RM Length L Ch R = 1 ,35225   ,526,526,526
BEGIN DESCRIPTION:
Stink Creek 66.1
END DESCRIPTION:
XS GIS Cut Line= 4
      1441364.21      6858355.19      1441570.99      6858301.19
       1441776.1      6858157.58      1442124.24      6857741.78
#Sta/Elev= 30
  4535.9 2040.59  4791.1 2040.31  4818.9 2034.64  4848.6 2031.15  4962.2 2030.03
  5005.9 2027.02  5006.4 2026.52  5019.2 2027.02  5059.9 2027.93  5084.1 2028.09
  5098.4 2032.14  5104.9 2031.41  5112.7 2033.19  5119.2 2031.42    5127    2033
  5133.5 2030.93  5141.3 2031.91  5162.2  2029.2  5197.3 2029.82  5211.6 2033.53
  5275.4 2034.72  5297.5 2034.18    5304 2032.43  5318.3 2033.67  5339.1 2031.44
  5353.4 2036.38  5361.2 2037.21  5453.6    2040  5517.4 2051.26  5542.3  2051.4
#Mann= 5 ,-1 , 0
  4535.9     .07       0  4962.2    .033       0  5005.9    .033       0
  5019.2    .033       0  5059.9     .07       0
Bank Sta=5005.9,5019.2
XS Rating Curve= 0 ,0
Exp/Cntr=0.3,0.1

Type RM Length L Ch R = 1 ,34699   ,69,69,69
BEGIN DESCRIPTION:
Stink Creek 66.0
END DESCRIPTION:
XS GIS Cut Line= 3
      1441360.77      6858369.09      1441955.68      6858532.34
      1443315.42       6858890.4
#Sta/Elev= 30
  4383.1 2040.33  4583.1  2038.4  4615.6 2037.79  4657.1 2035.04  4750.4  2032.9
  4791.9 2033.25  4810.5 2030.36  4815.7 2030.71  4850.1 2024.78  4855.3 2025.66
  4883.8 2025.06  4916.3 2025.07  4937.1 2023.54  5095.9 2022.87  5096.4 2022.37
  5109.6 2022.87  5197.2 2023.12  5235.1 2030.69  5240.3 2029.92  5275.4 2035.21
  5315.7 2034.52  5350.9 2036.36  5405.6 2035.97  5582.8 2035.26  5710.4 2035.57
  5836.9 2037.16  5864.6 2035.13    5897 2035.26  6373.3 2037.69  6406.1 2043.03
#Mann= 9 ,-1 , 0
  4383.1     .07       0  4883.8     .16       0  5095.9     .07       0
  5109.6     .16       0  5197.2     .07       0  5405.6     .16       0
  5582.8     .07       0  5710.4     .16       0    5897     .07       0
Bank Sta=5095.9,5109.6
XS Rating Curve= 0 ,0
Exp/Cntr=0.3,0.1

Type RM Length L Ch R = 1 ,34630   ,130,130,130
BEGIN DESCRIPTION:
Stink Creek 65.1
END DESCRIPTION:
XS GIS Cut Line= 6
       1441202.3      6858374.38      1441436.85      6858408.61
      1441819.39      6858571.34      1442056.81      6858632.28
      1442216.72      6858759.13      1443290.75      6858911.98
#Sta/Elev= 30
  4207.8 2041.24  4618.5 2035.95    4728 2038.69  4857.1 2037.76  4870.3  2039.3
  4915.4 2035.91  4920.5 2038.13  4948.2 2038.55  5102.6 2036.55  5108.9 2038.42
  5164.2 2038.53  5179.7 2038.38  5186.6 2035.82  5193.8 2038.06  5200.8 2034.79
    5208 2037.88  5214.9 2034.58  5222.1 2037.75  5229.1 2035.01  5236.3 2037.96
  5265.6  2038.3  5333.7 2033.99  5334.2 2033.49  5347.4 2033.99  5478.2 2034.76
  5604.6 2034.59  5742.2 2035.08  5818.7  2034.9  6374.4 2037.81  6399.9 2042.85
#Mann= 10 ,-1 , 0
  4207.8     .07       0  4857.1     .16       0  5164.2     .07       0
  5333.7     .07       0  5347.4     .07       0  5478.2    .035       0
  5604.6     .07       0  5742.2     .16       0  5818.7     .07       0
  6374.4     .16       0
Bank Sta=5333.7,5347.4
XS Rating Curve= 0 ,0
Exp/Cntr=0.3,0.1

Type RM Length L Ch R = 1 ,34500   ,500,500,500
BEGIN DESCRIPTION:
Stink Creek 65.0
END DESCRIPTION:
XS GIS Cut Line= 3
      1441294.27      6858609.01      1441922.93      6858720.65
      1443245.97      6858957.67
#Sta/Elev= 30
  4361.5 2039.86    4738 2032.14  4784.2 2033.91  4838.2  2029.8  4879.9 2029.25
  4910.7 2030.09  4941.2  2024.7  5003.6 2024.01  5010.2 2021.62  5015.3  2021.7
  5015.6 2019.14  5016.1 2018.64  5029.3 2019.14  5032.6 2022.14  5042.7  2023.5
  5093.5 2025.33  5134.2 2028.81  5168.7  2028.8  5215.4 2032.98  5235.4 2037.15
  5240.5 2034.87  5276.4 2038.54  5337.4 2034.34  5468.9 2034.06  5637.7 2034.41
  5727.3 2034.85  5764.8 2034.79  6199.1 2036.49  6317.7 2037.66  6344.1 2042.72
#Mann= 10 ,-1 , 0
  4361.5     .07       0  4879.9     .16       0  5015.6     .07       0
  5029.3     .16       0  5168.7     .07       0  5468.9    .035       0
  5637.7     .07       0  5727.3     .16       0  5764.8     .07       0
  6199.1     .16       0
Bank Sta=5015.6,5029.3
XS Rating Curve= 0 ,0
Exp/Cntr=0.3,0.1

Type RM Length L Ch R = 1 ,34000   ,500,500,500
BEGIN DESCRIPTION:
Stink Creek 64.0
END DESCRIPTION:
XS GIS Cut Line= 3
      1441264.33      6859110.77      1441708.53      6859079.51
      1443214.52      6858992.51
#Sta/Elev= 30
  4554.7 2045.48  4612.7 2045.03  4735.8 2043.44  4804.4 2039.38  4809.4 2040.48
  4865.9 2035.39  4950.8    2029  4966.4 2023.82    5000 2020.75  5009.6 2015.22
  5010.1 2014.72  5023.4 2015.22  5026.5 2016.76  5047.7 2019.59  5106.7 2021.58
  5112.3 2024.16  5117.3  2022.6  5284.1 2029.48  5357.1 2031.17  5784.6 2033.01
  5959.3 2032.79  6018.2 2032.18  6048.2 2033.67  6098.3 2033.11  6418.8 2038.18
  6458.9  2037.7  6478.9 2038.92    6497 2042.51    6502 2040.48  6508.5 2042.37
#Mann= 8 ,-1 , 0
  4554.7     .16       0  4612.7     .07       0  4865.9     .16       0
  5009.6     .07       0  5023.4     .16       0  5047.7     .07       0
  5784.6    .035       0  5959.3     .07       0
Bank Sta=5009.6,5023.4
XS Rating Curve= 0 ,0
Exp/Cntr=0.3,0.1

Type RM Length L Ch R = 1 ,33500   ,500,500,500
BEGIN DESCRIPTION:
Stink Creek 63.0
END DESCRIPTION:
XS GIS Cut Line= 3
      1441044.47      6859356.77      1441651.55      6859441.06
      1442798.49      6859358.55
#Sta/Elev= 30
  4387.1 2045.54  4417.9 2044.68  4478.5 2039.54  4629.9 2033.03  4831.9    2026
  4895.3 2026.52  4932.8 2023.04  4939.6  2020.8  4944.7 2021.71    4953 2020.82
  4973.2 2013.37  5006.6 2013.34  5007.1 2012.84  5020.4 2013.34  5073.6 2018.96
  5083.7 2021.31  5115.6 2021.55  5153.8 2025.66  5264.1 2028.41  5454.6 2028.21
  5504.8 2026.24  5574.9 2031.42    5605 2029.28  5705.3 2030.39  5755.4 2028.69
  5785.5 2030.47  5825.3 2030.64  6084.1 2033.03  6116.3 2033.36  6149.9 2036.96
#Mann= 6 ,-1 , 0
  4387.1     .07       0  4895.3     .16       0  5006.6     .07       0
  5020.4     .16       0  5825.3    .035       0  6084.1     .07       0
Bank Sta=5006.6,5020.4
XS Rating Curve= 0 ,0
Exp/Cntr=0.3,0.1

Type RM Length L Ch R = 1 ,33000   ,500,500,500
BEGIN DESCRIPTION:
Stink Creek 62.0
END DESCRIPTION:
XS GIS Cut Line= 3
      1440633.59      6859587.71      1441504.95      6859867.58
      1441954.57      6859586.96
#Sta/Elev= 30
  4084.8 2041.23  4222.8 2037.78  4235.7 2036.78  4460.5 2035.22  4548.4  2030.9
  4579.9 2030.35  4754.7 2023.11    4851 2022.53  4856.2 2023.57  4883.1 2020.53
  4888.4 2020.92  4913.4 2017.61  4926.5 2015.93  4947.3 2015.21  4952.6  2016.8
  4990.4 2011.13  4990.9 2010.63  5004.3 2011.13  5007.3 2014.51  5013.2 2013.88
  5022.6 2017.39  5028.5 2016.52  5035.4 2020.02  5043.9 2020.67  5049.8 2018.98
    5059  2018.8  5065.1 2020.55  5086.3 2022.37  5137.8 2023.93    5530 2026.47
#Mann= 5 ,-1 , 0
  4084.8     .07       0  4913.4     .16       0  4990.4     .07       0
  5004.3     .16       0  5137.8     .07       0
Bank Sta=4990.4,5004.3
XS Rating Curve= 0 ,0
Exp/Cntr=0.3,0.1

Type RM Length L Ch R = 1 ,32500   ,311,311,311
BEGIN DESCRIPTION:
Stink Creek 61.0
END DESCRIPTION:
XS GIS Cut Line= 3
      1440216.61      6861525.83      1441555.29      6860351.44
      1442355.29      6859645.25
#Sta/Elev= 30
  3219.2 2021.56  3239.5 2021.02  3577.6 2020.33  3918.2 2016.34  4132.4 2017.27
  4190.1 2018.25  4321.5 2020.53  4527.5  2018.4  4945.9 2018.82  4973.5 2017.15
  4981.1 2011.46  4988.1 2008.81  4988.6 2008.31  5002.4 2008.81  5009.5 2012.84
  5066.3 2012.05  5101.5 2018.73  5108.2 2018.21  5115.8 2014.04    5130 2009.99
  5158.4 2017.93  5214.4 2020.18  5426.9 2021.51  5477.2 2019.03  5491.4    2021
  5512.3 2020.07    5555 2022.39  5639.9 2023.37  5675.4 2021.94  6067.1  2029.1
#Mann= 6 ,-1 , 0
  3219.2    .045       0  3239.5     .07       0  4132.4    .035       0
  4190.1     .07       0  4988.1     .07       0  5002.4     .07       0
Bank Sta=4988.1,5002.4
XS Rating Curve= 0 ,0
Exp/Cntr=0.3,0.1

Type RM Length L Ch R = 1 ,32189   ,2265,2265,2265
BEGIN DESCRIPTION:
Stink Creek 60.0
END DESCRIPTION:
XS GIS Cut Line= 3
      1440399.83      6861622.08        1441555.      6860662.56
      1442498.57      6859862.03
#Sta/Elev= 30
  3498.3 2019.77  3668.3 2015.83  3810.2 2017.24  3824.5 2012.92  3980.8 2008.83
  4264.6 2009.35  4293.3 2014.48  4299.8 2012.14  4321.9 2015.48  4328.4 2012.41
  4336.2 2015.19  4342.7 2011.43  4357.1 2016.25  4406.5 2013.61  4414.4 2017.03
  4420.9 2013.41    4428 2017.29  4478.2 2017.96  4675.1 2016.04  4946.9 2017.11
    4961  2016.3  4974.3 2011.12  4974.9 2007.11  4975.4 2006.61  4989.3 2007.11
  5095.2 2017.26  5201.8 2012.24  5230.3 2016.66  5336.9 2020.63  6237.4 2031.18
#Mann= 4 ,-1 , 0
  3498.3     .07       0  4675.1    .035       0  4974.9    .035       0
  4989.3    .035       0
Bank Sta=4974.9,4989.3
XS Rating Curve= 0 ,0
Exp/Cntr=0.3,0.1

Type RM Length L Ch R = 1 ,29924   ,424,424,424
BEGIN DESCRIPTION:
Stink Creek 58.0
END DESCRIPTION:
XS GIS Cut Line= 3
      1440410.83      6861680.61       1441097.5      6861791.13
      1442570.53      6861723.03
#Sta/Elev= 30
  4304.5 2017.29  4373.9 2015.83  4470.8 2013.87  4512.3 2012.14  4551.8 2011.95
  4606.5 2009.71    4735 2006.42  4794.9 2005.71  4821.6 2002.21  4826.7 2002.64
  4865.8  1999.8  4875.9 2000.58    4957 1999.26  4967.1 2000.18    5000 1997.37
  5000.2 1996.43  5000.7 1995.93  5014.9 1996.43  5017.5 1999.64  5027.5 2005.59
  5037.5 2006.99  5209.8 2008.82  5231.6 2008.93  5393.5 2009.92  5441.5 2010.07
  5688.2 2010.46  5718.3 2011.62  6028.6 2013.02  6238.8  2016.3  6474.6 2021.75
#Mann= 10 ,-1 , 0
  4304.5     .07       0  4373.9    .035       0  4606.5     .07       0
    4735     .16       0  5000.2     .07       0  5014.9     .16       0
  5209.8     .16       0  5231.6     .07       0  5393.5     .16       0
  5441.5     .07       0
Bank Sta=5000.2,5014.9
XS Rating Curve= 0 ,0
Exp/Cntr=0.3,0.1

Type RM Length L Ch R = 1 ,29500   ,321,321,321
BEGIN DESCRIPTION:
Stink Creek 57.0
END DESCRIPTION:
XS GIS Cut Line= 3
      1440482.37      6862153.13      1440955.04      6862158.66
      1441904.96      6862337.99
#Sta/Elev= 30
  4527.3 2012.38  4629.9 2012.93  4709.9  2010.9  4789.9 2006.27  4905.7 2003.61
    4960 2000.36    4980 2001.62    4990 1999.14  4997.5 1994.31  5002.5 1994.31
  5002.8 1991.69  5003.3 1991.19  5017.5 1991.69  5019.3 1993.97  5024.4 1994.05
  5030.5 1997.42  5081.5 2003.68  5122.1 2003.18  5401.3 2005.12  5511.2 2003.36
  5578.9 2003.55  5621.1 2003.69  5641.1 2006.06  5661.4 2006.11    5753 2012.64
  5830.7 2013.12  5844.6 2013.97  5883.1  2013.4  5944.2 2014.09  5966.7 2014.13
#Mann= 7 ,-1 , 0
  4527.3     .07       0  4905.7     .16       0  5002.8     .07       0
  5017.5     .16       0  5081.5     .07       0  5578.9     .16       0
  5944.2     .07       0
Bank Sta=5002.8,5017.5
XS Rating Curve= 0 ,0
Exp/Cntr=0.3,0.1

Type RM Length L Ch R = 1 ,29179   ,882,882,882
BEGIN DESCRIPTION:
Stink Creek 56.0
END DESCRIPTION:
XS GIS Cut Line= 3
      1439596.09      6862480.89      1440904.68      6862463.29
      1441805.02        6862438.
#Sta/Elev= 30
  3691.3 2010.27  3740.2 2005.29  3782.4 2004.44    3971 2003.22  4150.2 2002.23
  4330.3 2003.15  4390.3 2005.06  4530.3 2006.14  4920.3 2003.33  4950.3    2001
  4960.3 1999.06  4970.3 1994.88    4973 1990.02  4973.5 1989.52  4987.7 1990.02
  4990.3 1992.45  4997.7 1994.81  5047.9 1998.23  5070.4 2000.03  5140.4 2001.44
  5200.4 2000.67  5245.3 2001.92  5590.6 2001.84  5620.6 2002.18  5630.6 2003.43
  5670.6 2003.11  5691.7 2004.79  5831.1 2012.64  5870.7 2015.87  5900.7 2015.65
#Mann= 9 ,-1 , 0
  3691.3     .07       0  3782.4    .035       0    3971     .07       0
    4973     .07       0  4987.7     .07       0  5047.9     .16       0
  5245.3     .07       0  5691.7     .16       0  5831.1     .07       0
Bank Sta=4973,4987.7
XS Rating Curve= 0 ,0
Exp/Cntr=0.3,0.1

Type RM Length L Ch R = 1 ,28297   ,218,218,218
BEGIN DESCRIPTION:
Stink Creek 55.0
END DESCRIPTION:
XS GIS Cut Line= 3
      1439506.67       6862529.1      1441545.01        6862928.
        1442055.      6863001.03
#Sta/Elev= 30
    2923 2010.65  2996.5 2009.78  3034.4  2006.4  3074.1 2003.88  3183.4 2001.74
  3259.2  2002.6    3390 2001.11  3940.3 2000.82  4164.4 2001.79  4500.5 1999.54
  4592.4  1998.5  4633.2 1996.62  4684.1 1998.55  4735.1 1998.36  4866.1 1996.64
  4917.6 1992.87  4974.3 1991.84  5002.7  1987.6  5003.2  1987.1  5017.5  1987.6
  5030.3 1992.98  5035.3  1989.9  5050.5  1992.8  5080.8 1993.07  5100.9 1995.55
  5131.3 2003.64  5141.4 2004.61  5385.8 2010.64  5485.4 2014.15  5515.2 2015.23
#Mann= 7 ,-1 , 0
    2923     .07       0  3034.4    .035       0  3183.4     .07       0
  5002.7     .07       0  5017.5     .07       0  5385.8    .035       0
  5485.4     .07       0
Bank Sta=5002.7,5017.5
XS Rating Curve= 0 ,0
Exp/Cntr=0.3,0.1

Type RM Length L Ch R = 1 ,28079   ,579,579,579
BEGIN DESCRIPTION:
Stink Creek 54.0
END DESCRIPTION:
XS GIS Cut Line= 3
      1439576.81      6862647.43      1441654.67      6863103.42
      1442070.21      6863149.61
#Sta/Elev= 30
  2872.7 2007.03  2973.2 2001.17  3157.5 2000.01  3259.9 1997.96  3300.8 1999.75
  3792.3    1999    3823 1999.86  3878.8 1999.17    3997 2000.55  4181.3 2000.35
  4205.9 2001.08  4300.8 2000.13  4467.7 1998.03  4652.2 1996.86  4784.8 1994.86
  4811.2 1993.13  4867.2 1991.56  4971.3 1991.27  4979.9 1991.39  4989.2 1985.86
  4989.7 1985.36    5004 1985.86  5070.8 1989.26  5080.8  1990.5  5086.3 1994.13
  5091.3 1991.94    5111 2003.05  5121.1 2004.78  5211.6 2008.22  5418.1 2014.03
#Mann= 7 ,-1 , 0
  2872.7    .035       0  4300.8     .07       0  4467.7    .035       0
  4784.8     .07       0  4971.3    .035       0  4989.2    .035       0
    5004    .035       0
Bank Sta=4989.2,5004
XS Rating Curve= 0 ,0
Exp/Cntr=0.3,0.1

Type RM Length L Ch R = 1 ,27500   ,500,500,500
BEGIN DESCRIPTION:
Stink Creek 53.0
END DESCRIPTION:
XS GIS Cut Line= 3
      1439564.53      6862704.76      1441506.18      6863500.29
      1441851.27      6863827.27
#Sta/Elev= 30
  2901.7 2005.92  3033.1 2000.22  3226.4 1999.03  3294.7 1996.94  3342.7 1998.42
  3559.1 1997.72  3859.4 1998.14  4453.1 1997.73    4864 1992.43  4981.6 1989.82
  4996.7 1983.27  5011.3 1981.67  5011.8 1981.17  5026.2 1981.67  5032.9 1987.72
    5054 1987.75  5103.7 1992.39  5152.1 1992.88  5259.4 1995.28  5280.5 1996.74
  5308.8 2001.29  5329.8 2006.34  5337.1 2006.18    5344 2008.03  5351.3 2006.37
  5365.4 2007.07  5372.3 2009.03  5386.5 2010.19  5393.7 2009.09  5475.4 2012.76
#Mann= 7 ,-1 , 0
  2901.7     .07       0  3559.1    .035       0  3859.4     .07       0
    4864     .16       0  5011.3     .07       0  5026.2     .16       0
  5152.1     .07       0
Bank Sta=5011.3,5026.2
XS Rating Curve= 0 ,0
Exp/Cntr=0.3,0.1

Type RM Length L Ch R = 1 ,27000   ,624,624,624
BEGIN DESCRIPTION:
Stink Creek 52.0
END DESCRIPTION:
XS GIS Cut Line= 3
      1439523.48      6862749.62      1441239.92      6863903.08
      1441524.08      6864081.06
#Sta/Elev= 30
    2932 2006.52  2934.5 2006.52    3032 2000.75  3115.6 1999.56  3282.7 1997.91
    3371  1995.9  3524.7 1996.81    3644 1995.98    4214 1994.95  4271.2 1995.78
    4337 1993.96    4424 1993.92    4517 1992.02  4921.8 1988.85    4949  1986.2
  4957.9 1983.81  4962.6 1979.16  4963.1 1978.66  4977.5 1979.16    4985 1982.05
  4999.9 1984.93  5057.7 1988.63  5073.1 1988.11  5209.8 1996.67  5238.3 2001.36
  5261.6 2003.35  5282.9  2003.6  5298.2 2006.25  5319.4 2007.72  5335.3 2007.34
#Mann= 9 ,-1 , 0
    2932    .035       0  2934.5     .07       0  3115.6    .035       0
  3282.7     .07       0  3524.7    .035       0    3644     .07       0
  4962.6     .07       0  4977.5     .07       0  5238.3    .035       0
Bank Sta=4962.6,4977.5
XS Rating Curve= 0 ,0
Exp/Cntr=0.3,0.1

Type RM Length L Ch R = 1 ,26376   ,553,553,553
BEGIN DESCRIPTION:
Stink Creek 51.0
END DESCRIPTION:
XS GIS Cut Line= 3
      1439308.26       6862599.5      1440784.95      6864187.65
      1441091.03       6864350.7
#Sta/Elev= 30
  2831.4  2015.3  2856.6 2010.42  2877.6 2008.29  2936.5  2008.6  2957.1 2007.54
  3098.8 2005.85  3132.1 2005.13    3182 2001.31  3242.1 2000.09  3641.7 1994.73
  3787.2 1995.37  4526.1 1991.68  4653.6 1987.99  4781.2 1986.04  4941.7 1985.78
  4964.9 1984.46    4979  1977.6  4985.7 1976.19  4986.2 1975.69  5000.7 1976.19
  5014.2 1983.67  5045.4 1985.04  5116.6 1983.81  5162.3 1981.92  5184.3 1982.42
  5206.2  1987.2    5238 1989.86  5266.5 1994.73    5303 1995.04  5346.8 2000.68
#Mann= 11 ,-1 , 0
  2831.4    .035       0  2936.5     .07       0  2957.1    .035       0
  3098.8     .07       0  3242.1    .035       0  3787.2     .07       0
  4941.7     .16       0  4985.7     .07       0  5000.7     .16       0
  5116.6    .035       0    5303    .063       0
Bank Sta=4985.7,5000.7
XS Rating Curve= 0 ,0
Exp/Cntr=0.3,0.1

Type RM Length L Ch R = 1 ,25823   ,323,323,323
BEGIN DESCRIPTION:
Stink Creek 50.0
END DESCRIPTION:
XS GIS Cut Line= 3
      1439423.43      6864862.98      1440508.77      6864536.43
      1441185.63        6864423.
#Sta/Elev= 30
  3866.6 2000.56  3930.8  1999.1  4024.9 1994.76  4048.6 1992.72  4202.4 1988.83
  4369.5 1982.85  4400.8  1983.2  4424.4  1981.8  4457.4 1983.75  4463.5 1983.05
  4495.7 1984.33  4745.4 1985.47  4841.5 1984.61  4973.6 1980.41    5000 1977.94
  5007.9 1975.61  5008.4 1975.11  5024.3 1975.61  5076.7 1977.01  5087.4 1980.25
  5117.9 1982.77  5239.5 1982.76  5324.5  1985.6  5371.3 1985.79  5380.1 1986.82
    5391 1985.99  5440.8 1990.51  5592.7 1994.78  5683.4 1999.57  5686.3 1998.39
#Mann= 6 ,-1 , 0
  3866.6    .063       0  4048.6    .035       0  5007.9    .035       0
  5024.3    .035       0    5391    .063       0  5592.7    .094       0
Bank Sta=5007.9,5024.3
XS Rating Curve= 0 ,0
Exp/Cntr=0.3,0.1

Type RM Length L Ch R = 1 ,25500   ,500,500,500
BEGIN DESCRIPTION:
Stink Creek 49.0
END DESCRIPTION:
XS GIS Cut Line= 3
      1440325.37      6864919.28      1441126.82      6864659.45
      1441270.42       6864689.4
#Sta/Elev= 30
  4704.5 1982.69  4823.6 1981.84  4914.3 1979.78  4956.8 1979.89  4983.5 1978.88
  4998.5 1975.33  5000.8 1973.84  5001.3 1973.34  5017.2 1973.84  5052.7 1975.11
  5084.7 1978.57  5111.4  1977.6  5116.7  1979.2  5135.1  1978.3  5148.6 1979.84
  5166.7 1979.93  5239.3 1983.17  5276.6 1983.22  5303.3 1984.66  5386.8 1986.23
  5504.8 1990.16  5524.1 1990.73  5532.4 1991.23  5537.7  1992.5  5562.4 1993.59
  5567.5 1992.42  5612.5 1994.68  5617.6 1993.37  5648.1 1994.43  5693.7 1996.13
#Mann= 6 ,-1 , 0
  4704.5    .035       0  5000.8    .035       0  5017.2    .035       0
  5386.8    .063       0  5504.8    .035       0  5648.1     .07       0
Bank Sta=5000.8,5017.2
XS Rating Curve= 0 ,0
Exp/Cntr=0.3,0.1

Type RM Length L Ch R = 1 ,25000   ,500,500,500
BEGIN DESCRIPTION:
Stink Creek 48.0
END DESCRIPTION:
XS GIS Cut Line= 3
      1440313.59      6865171.54      1440872.09      6865205.09
      1441505.01      6864787.99
#Sta/Elev= 30
  4440.5 1981.23  4605.4 1980.96  4652.3 1981.38  4704.4 1979.49  4708.4 1979.46
  4902.4 1976.13  4922.8 1970.83  4924.6 1968.52  4925.1 1968.02    4941 1968.52
  4961.5 1972.85  4966.5 1969.82  4972.9 1969.18    4999 1972.58  5006.6 1976.22
  5027.7 1976.68  5051.4 1971.85  5072.9 1970.54  5130.1 1969.66  5223.5 1970.84
  5295.7 1974.41  5302.9 1975.09  5310.8 1978.26  5316.8 1977.11  5325.9 1980.01
  5331.9 1978.43  5346.9 1983.16  5383.1 1985.76  5749.8 2002.42    5758 2002.71
#Mann= 8 ,-1 , 0
  4440.5     .07       0  4605.4    .035       0  4704.4     .07       0
  4708.4    .035       0  4902.4     .07       0  4924.6     .07       0
    4941     .07       0  5749.8    .035       0
Bank Sta=4924.6,4941
XS Rating Curve= 0 ,0
Exp/Cntr=0.3,0.1

Type RM Length L Ch R = 1 ,24500   ,500,500,500
BEGIN DESCRIPTION:
Stink Creek 47.0
END DESCRIPTION:
XS GIS Cut Line= 3
      1440543.89      6865270.65      1441116.87      6865550.09
      1441505.02      6865037.97
#Sta/Elev= 30
  4362.5 1979.52  4396.1 1979.38  4396.2 1979.38  4613.5  1978.4  4632.7 1978.15
  4728.7 1977.13  4802.3  1977.2  4818.1 1976.32  4920.5 1974.23  4937.5 1968.18
    4943 1967.61  4953.4 1971.95    4960 1973.54  4965.6 1970.91  4975.7 1970.16
  4979.8 1967.57  4980.3 1967.07  4996.3 1967.57  5015.2 1969.45  5021.6 1972.76
  5027.9 1973.45  5228.5    1977    5265 1978.43  5285.8 1980.43  5441.8 1989.46
    5492 1990.54  5506.3 1992.05  5514.6 1991.54  5535.4 1993.13  5642.6 1996.95
#Mann= 9 ,-1 , 0
  4362.5     .07       0  4396.1    .035       0  4396.2     .07       0
  4613.5    .035       0  4632.7     .07       0  4728.7    .035       0
  4818.1     .07       0  4979.8     .07       0  4996.3     .07       0
Bank Sta=4979.8,4996.3
XS Rating Curve= 0 ,0
Exp/Cntr=0.3,0.1

Type RM Length L Ch R = 1 ,24000   ,500,500,500
BEGIN DESCRIPTION:
Stink Creek 46.0
END DESCRIPTION:
XS GIS Cut Line= 4
      1440862.51      6865639.47      1441048.43      6866012.15
      1441315.71      6865938.21      1441704.97      6865438.03
#Sta/Elev= 30
  4306.2 1976.57  4843.6 1973.53  4864.4 1971.99  4869.5 1970.52  4874.8 1965.48
  4876.9 1964.81  4877.4 1964.31  4893.4 1964.81  4895.5 1967.25    4909 1971.59
  4916.3 1971.66  4943.4 1966.05  4957.8 1970.04  4988.9 1971.43    4997 1969.16
  5003.3 1969.16  5013.1 1971.21  5035.7 1969.85  5085.5 1971.37  5106.3 1973.86
  5127.1 1970.41  5135.3 1972.07  5141.6 1970.63    5185 1973.37  5285.1 1976.45
  5363.3 1980.23  5469.2 1988.57  5506.3 1988.19  5527.1 1990.03  5633.8 1993.38
#Mann= 4 ,-1 , 0
  4306.2     .07       0  4876.9     .07       0  4893.4     .07       0
  5285.1     .07       0
Bank Sta=4876.9,4893.4
XS Rating Curve= 0 ,0
Exp/Cntr=0.3,0.1

Type RM Length L Ch R = 1 ,23500   ,500,500,500
BEGIN DESCRIPTION:
Stink Creek 45.0
END DESCRIPTION:
XS GIS Cut Line= 3
        1439455.        6865188.      1441314.48      6866280.17
      1441704.96      6866088.02
#Sta/Elev= 30
  2843.5 2002.69  2881.1 1999.01  2915.7  1998.9  3041.1 1992.61  3214.6 1984.53
    3326 1981.75  3547.4 1979.28  3763.6 1976.41  3779.2 1977.97    3785 1976.12
  3871.4 1975.12  4115.2 1972.31  4195.3 1973.23  4318.3 1971.34  4392.6  1973.3
  4685.7 1973.47  4995.2 1968.91  5016.8 1968.69  5036.9 1962.84  5037.4 1962.34
  5053.4 1962.84  5061.7 1963.45  5067.5 1967.62  5092.3 1967.66  5190.1 1972.42
  5308.9 1980.39  5336.9 1981.08  5381.9 1983.93  5398.8 1986.76  5435.2 1988.43
#Mann= 9 ,-1 , 0
  2843.5    .063       0  2881.1    .035       0  3041.1     .07       0
  3547.4     .16       0  3871.4     .07       0  4995.2     .16       0
  5036.9     .07       0  5053.4     .16       0  5092.3     .07       0
Bank Sta=5036.9,5053.4
XS Rating Curve= 0 ,0
Exp/Cntr=0.3,0.1

Type RM Length L Ch R = 1 ,23000   ,500,500,500
BEGIN DESCRIPTION:
Stink Creek 44.0
END DESCRIPTION:
XS GIS Cut Line= 3
      1439405.02      6865238.01      1441098.49       6866646.1
      1441755.02      6866838.01
#Sta/Elev= 30
  2797.6 2002.49    2822  2001.8  2903.7 2000.75  2950.7 1997.67  3024.8 1991.14
  3196.9 1984.55    3242 1983.83  3380.2 1982.12  3386.7 1983.67  3415.4 1980.67
  4000.3 1974.94  4007.7 1974.84  4158.9 1973.17  4247.6 1971.68  4290.7 1971.32
  4413.2 1969.47  4934.8 1965.92  4970.3 1967.27  4997.6 1961.82  5006.8 1961.96
  5008.9 1959.47  5009.4 1958.97  5025.5 1959.47  5028.7 1964.47    5038 1965.84
  5227.7 1969.37  5329.8  1979.4    5361 1976.56  5417.4 1979.35    5684 1985.65
#Mann= 16 ,-1 , 0
  2797.6    .063       0    2822    .035       0  2950.7     .07       0
  3196.9     .16       0    3242     .07       0  4000.3    .035       0
  4007.7     .07       0  4158.9    .035       0  4247.6     .07       0
  4290.7    .035       0  4413.2     .07       0  4970.3     .16       0
  5008.9     .07       0  5025.5     .16       0  5227.7     .07       0
  5417.4    .045       0
Bank Sta=5008.9,5025.5
XS Rating Curve= 0 ,0
Exp/Cntr=0.3,0.1

Type RM Length L Ch R = 1 ,22500   ,500,500,500
BEGIN DESCRIPTION:
Stink Creek 43.0
END DESCRIPTION:
XS GIS Cut Line= 3
      1439354.96      6865787.97      1440762.29      6866880.79
      1441704.96        6866938.
#Sta/Elev= 30
  3218.2 1997.44  3275.3 1996.68  3310.6 1997.54  3361.7 1993.54  3424.6 1988.56
  3525.2 1984.43  3681.6 1979.83  3724.7 1979.92  3994.8 1974.65  4280.8 1971.73
  4672.7 1969.26    4851 1965.05  4857.3 1963.96  4907.1 1963.16    4960 1963.94
  4971.4 1963.31  4977.6 1957.79  4978.1 1957.29  4994.2 1957.79  4998.5 1962.68
  5063.4 1963.38  5206.1 1964.07  5423.4 1964.75  5535.2 1969.33  5643.9 1978.69
  5673.9 1978.26  5698.5 1979.92  5744.1 1982.84  5774.1 1982.45  5944.4 1986.93
#Mann= 10 ,-1 , 0
  3218.2    .035       0  3361.7     .16       0  3525.2     .07       0
    4960     .16       0  4977.6     .07       0  4994.2     .16       0
  5063.4     .07       0  5206.1     .16       0  5423.4     .07       0
  5698.5    .045       0
Bank Sta=4977.6,4994.2
XS Rating Curve= 0 ,0
Exp/Cntr=0.3,0.1

Type RM Length L Ch R = 1 ,22000   ,500,500,500
BEGIN DESCRIPTION:
Stink Creek 42.0
END DESCRIPTION:
XS GIS Cut Line= 3
      1439504.97      6866537.98      1440749.08      6867341.63
      1441705.01        6867088.
#Sta/Elev= 30
  3518.9 1987.64  3583.9 1986.65  3620.2 1984.09  3755.9 1979.83  3891.6 1975.74
  4025.3 1972.45  4155.3 1971.41  4191.6 1969.92  4481.9 1965.13    4813 1961.53
  4929.2 1962.35  4944.4 1960.65  4959.4 1961.86  4965.5 1958.09  4971.5 1957.67
  4972.3 1955.85  4972.8 1955.35  4989.1 1955.85  4994.6 1960.59  5006.1 1961.22
  5268.8 1963.37  5410.9 1967.98  5620.1 1975.85  5668.3 1979.07  5685.9 1978.19
  5700.5  1978.2  5730.3 1981.32  5775.7 1981.21  5926.1 1986.48    5989 1987.53
#Mann= 8 ,-1 , 0
  3518.9     .07       0  3755.9    .035       0  3891.6     .07       0
    4813     .16       0  4972.3     .07       0  4989.1     .16       0
  5410.9     .07       0  5685.9    .045       0
Bank Sta=4972.3,4989.1
XS Rating Curve= 0 ,0
Exp/Cntr=0.3,0.1

Type RM Length L Ch R = 1 ,21500   ,500,500,500
BEGIN DESCRIPTION:
Stink Creek 41.0
END DESCRIPTION:
XS GIS Cut Line= 3
      1439669.52      6867463.52      1440512.87      6867645.69
      1441455.04      6867237.98
#Sta/Elev= 30
  4137.2  1982.1  4163.3 1979.99  4180.4 1977.16  4204.2 1976.78  4229.6  1975.7
  4234.9  1974.8  4278.9 1973.39  4347.4 1969.18  4429.3 1967.11  4465.7 1965.33
  4541.8 1963.77    4751 1962.39  4807.8 1961.25    4859 1961.63  4869.2 1960.74
  4895.3 1960.83  4930.6 1959.69  4937.8 1958.56    4951 1958.91  4973.3 1955.72
  4973.8 1955.22  4990.2 1955.72  4998.5 1959.76  5097.1 1959.55  5190.4 1958.37
  5616.1 1967.25  5958.6 1977.55    5983 1978.35  6004.8 1980.47  6026.6 1979.87
#Mann= 8 ,-1 , 0
  4137.2     .07       0  4895.3     .16       0  4973.3     .07       0
  4990.2     .16       0  5097.1     .07       0  5190.4     .16       0
  5616.1     .07       0  5958.6    .045       0
Bank Sta=4973.3,4990.2
XS Rating Curve= 0 ,0
Exp/Cntr=0.3,0.1

Type RM Length L Ch R = 1 ,21000   ,500,500,500
BEGIN DESCRIPTION:
Stink Creek 40.0
END DESCRIPTION:
XS GIS Cut Line= 4
      1439633.24      6867489.34      1440542.11      6867979.42
       1440854.2      6867907.29      1441504.96      6867788.01
#Sta/Elev= 30
  3647.1 1982.31  3651.9 1982.22    3671 1982.27  3714.8 1979.25  3742.4 1978.69
  3764.3 1975.86  3785.3 1974.56  3906.2 1969.74  3944.3 1967.33  4053.8  1964.2
  4126.3 1963.43  4163.3 1961.77    4349 1960.07    4666 1960.34  4861.2 1956.85
  4908.4  1956.6  4949.5 1957.75  4969.8 1956.65  4980.3 1954.19  4982.1 1952.93
  4982.6 1952.43    4999 1952.93    5000 1956.62    5025 1957.79  5131.3 1956.36
  5172.5 1957.27  5247.8 1960.01  5300.9 1964.08  5435.4 1971.49  5661.6 1979.19
#Mann= 8 ,-1 , 0
  3647.1     .07       0  3651.9    .035       0  3785.3     .07       0
  4861.2     .16       0  4982.1     .07       0    4999     .16       0
  5172.5     .07       0  5435.4    .045       0
Bank Sta=4982.1,4999
XS Rating Curve= 0 ,0
Exp/Cntr=0.3,0.1

Type RM Length L Ch R = 1 ,20500   ,500,500,500
BEGIN DESCRIPTION:
Stink Creek 39.0
END DESCRIPTION:
XS GIS Cut Line= 3
      1439554.99      6867487.99      1440964.96      6868278.79
        1441455.        6868038.
#Sta/Elev= 30
  3383.4 1982.61  3413.1 1983.71  3494.1 1981.48  3601.6 1975.26  3861.5 1963.92
    3970  1961.6  4207.3  1959.5  4461.8 1960.16  4635.3 1956.39  4764.1 1953.25
  4801.8 1954.77  4845.2 1953.47  4977.1 1955.22  4991.2 1954.78  4997.2 1952.74
  5013.8 1951.01  5014.3 1950.51  5030.8 1951.01  5066.9 1955.06    5234 1958.42
  5245.3  1959.5  5262.2 1967.77  5278.6 1969.11  5307.2 1962.76  5349.2 1962.91
  5374.6 1963.45    5390 1965.05  5402.7 1968.68  5425.2 1970.21    5546 1975.02
#Mann= 6 ,-1 , 0
  3383.4    .035       0  3601.6     .07       0  4635.3     .16       0
  5013.8     .07       0  5030.8     .16       0  5349.2     .07       0
Bank Sta=5013.8,5030.8
XS Rating Curve= 0 ,0
Exp/Cntr=0.3,0.1

Type RM Length L Ch R = 1 ,20000   ,1000,1000,1000
BEGIN DESCRIPTION:
Stink Creek 38.0
END DESCRIPTION:
XS GIS Cut Line= 3
      1439554.98      6867587.99      1440540.73      6868302.21
        1441705.        6868538.
#Sta/Elev= 30
  3782.7 1982.53  3832.1 1980.68    3855 1981.29  3869.2 1979.92  3905.3 1980.15
  3984.4  1975.9  4219.2 1963.57  4355.3 1959.92  4571.1 1958.83  4843.3 1959.34
    4950  1958.5  4986.8 1956.39  5014.6 1953.91  5036.7  1947.9  5037.2  1947.4
  5053.7  1947.9  5057.4 1953.24    5086  1951.7  5204.4 1953.32  5305.8 1952.64
  5330.8 1954.22  5351.3 1951.75  5371.7 1954.22  5392.1 1954.32  5422.7 1956.57
  5598.4 1962.46  5711.4  1965.3  5907.8 1972.88  6080.9 1979.21  6187.9 1982.46
#Mann= 8 ,-1 , 0
  3782.7    .035       0  3984.4     .07       0  4986.8     .16       0
  5036.7     .07       0  5053.7     .16       0  5598.4     .07       0
  5907.8    .035       0  6080.9    .045       0
Bank Sta=5036.7,5053.7
XS Rating Curve= 0 ,0
Exp/Cntr=0.3,0.1

Type RM Length L Ch R = 1 ,19000   ,500,500,500
BEGIN DESCRIPTION:
Stink Creek 37.0
END DESCRIPTION:
XS GIS Cut Line= 3
      1439504.98      6867687.99      1440741.57      6868801.58
      1441555.03      6868537.99
#Sta/Elev= 30
  3335.9 1979.94  3400.9 1977.97  3576.6 1973.39  3675.6  1968.4  3725.7 1964.37
  3838.5 1959.64  4001.5 1957.75  4398.3 1957.93  4624.8 1956.17  4837.1  1951.9
  4886.4 1952.28  4957.4 1948.13  5014.1 1948.28  5023.6 1946.91  5028.9 1948.47
  5037.2 1943.81  5037.7 1943.31  5054.2 1943.81  5055.6 1945.83  5060.9  1945.2
  5066.7 1948.12  5087.6  1949.8  5092.8 1947.67  5098.2 1951.63  5108.7 1952.84
  5130.1 1951.61  5156.8 1954.03  5320.2 1958.22  5709.2 1972.79  5855.1  1977.7
#Mann= 7 ,-1 , 0
  3335.9     .07       0  3400.9    .035       0  3576.6     .07       0
  5037.2     .07       0  5054.2     .07       0  5320.2     .07       0
  5709.2    .035       0
Bank Sta=5037.2,5054.2
XS Rating Curve= 0 ,0
Exp/Cntr=0.3,0.1

Type RM Length L Ch R = 1 ,18500   ,500,500,500
BEGIN DESCRIPTION:
Stink Creek 36.0
END DESCRIPTION:
XS GIS Cut Line= 3
      1439404.98      6867987.98      1440654.98      6869239.58
      1441304.98        6869288.
#Sta/Elev= 30
  3231.1 1976.37  3322.8 1971.29  3379.6  1969.5  3386.7 1967.41  3429.1 1967.01
  3457.4 1964.22  3510.7 1961.31  3662.5 1956.73  3846.3 1955.72  3888.7 1956.41
  3952.4 1955.41  4362.5 1955.87  4593.6 1954.46    4806 1952.68  4869.9 1952.32
    4914 1952.25  4921.1  1951.8  4928.2 1949.74  4962.4 1949.82  4996.1 1945.69
    5000 1945.58  5001.5 1941.95    5002 1941.45  5018.6 1941.95  5030.1 1946.34
  5077.2 1947.94  5183.1  1950.3  5310.6 1955.58  5461.3 1959.74  5651.8 1968.76
#Mann= 10 ,-1 , 0
  3231.1     .07       0  3322.8    .035       0  3510.7     .07       0
  4593.6    .035       0    4806    .045       0  4869.9     .07       0
  4996.1    .035       0  5001.5    .035       0  5018.6    .035       0
  5077.2     .07       0
Bank Sta=5001.5,5018.6
XS Rating Curve= 0 ,0
Exp/Cntr=0.3,0.1

Type RM Length L Ch R = 1 ,18000   ,500,500,500
BEGIN DESCRIPTION:
Stink Creek 35.0
END DESCRIPTION:
XS GIS Cut Line= 3
      1439404.98      6868137.97      1440655.55      6869707.72
      1441304.97      6869438.01
#Sta/Elev= 30
    2993 1970.15  3044.7 1968.12  3085.1 1966.95    3114 1963.32  3157.2 1962.73
  3250.6 1957.35  3413.4 1954.93  3640.9 1954.31  3847.5 1955.65  3976.2 1954.56
  4135.2 1952.99  4408.8 1952.15  4427.2 1952.08  4662.8 1950.94  4793.7 1949.51
  4808.4 1947.79  4936.4 1947.79  4985.3  1944.4  5002.4 1944.03  5012.5 1939.45
    5013 1938.95  5029.6 1939.45  5034.5 1941.63  5043.3 1942.05  5061.7 1946.12
  5107.7 1949.05  5393.6 1956.38  5510.7 1958.53  5666.6  1965.4  5703.2 1966.58
#Mann= 15 ,-1 , 0
    2993     .07       0  3044.7    .035       0  3250.6     .07       0
  3976.2    .035       0  4135.2    .045       0  4408.8     .07       0
  4427.2    .045       0  4662.8     .07       0  4793.7    .035       0
  4985.3     .07       0  5012.5     .07       0  5029.6     .07       0
  5034.5     .16       0  5393.6     .07       0  5666.6    .035       0
Bank Sta=5012.5,5029.6
XS Rating Curve= 0 ,0
Exp/Cntr=0.3,0.1

Type RM Length L Ch R = 1 ,17500   ,500,500,500
BEGIN DESCRIPTION:
Stink Creek 34.0
END DESCRIPTION:
XS GIS Cut Line= 3
      1439355.02      6868088.03      1440449.33      6870088.82
      1440448.81      6870252.52
#Sta/Elev= 30
  2719.5 1972.46  2868.7 1967.36  2934.3 1965.06    2940 1961.58  2947.4 1960.97
    2993 1960.49  3027.3 1957.36  3111.5 1955.58  3520.5 1954.58  3629.6 1953.04
  3758.6 1952.38  4193.4  1950.8  4196.1  1950.8  4309.4 1950.63  4387.6 1949.81
  4429.6 1949.46    4522 1949.14  4661.3 1947.94  4839.9 1945.14  4921.5 1946.25
  4953.5  1943.2  4959.4  1940.3  4979.1 1937.47  4979.6 1936.97  4996.3 1937.47
  5002.1 1938.53  5009.2 1942.33  5059.2 1951.61    5144 1952.04  5163.7 1951.99
#Mann= 16 ,-1 , 0
  2719.5     .07       0  2868.7    .035       0  3111.5     .07       0
  3520.5    .035       0  3629.6     .07       0  3758.6    .045       0
  4193.4     .07       0  4196.1    .045       0  4309.4     .07       0
  4387.6    .045       0  4429.6     .07       0    4522    .045       0
  4661.3     .07       0  4979.1     .07       0  4996.3     .07       0
    5144    .035       0
Bank Sta=4979.1,4996.3
XS Rating Curve= 0 ,0
Exp/Cntr=0.3,0.1

Type RM Length L Ch R = 1 ,17000   ,500,500,500
BEGIN DESCRIPTION:
Stink Creek 33.0
END DESCRIPTION:
XS GIS Cut Line= 3
      1439404.99      6868237.96      1440045.74      6870247.79
      1440155.01      6870338.01
#Sta/Elev= 30
  2890.5 1967.65  2920.8 1966.29    2985 1963.28  3016.5 1959.07  3099.9 1955.68
    3237 1954.17  3371.7 1954.22  3457.3 1954.03  3496.8 1952.33    3566 1952.08
    3765 1952.24  3801.8 1951.45  4269.1 1948.99  4376.9 1948.16  4506.9 1947.95
  4553.6 1946.73  4632.9 1946.84  4696.1 1945.43    4946 1943.83  4958.2 1944.08
  5006.8 1940.98  5021.2 1938.99  5026.9 1936.33  5027.4 1935.83  5044.1 1936.33
  5049.9 1941.82  5056.3 1942.59  5063.9 1944.95    5111 1946.58  5141.7 1946.82
#Mann= 13 ,-1 , 0
  2890.5     .07       0  2920.8    .035       0    3237     .07       0
  3371.7    .035       0    3566     .07       0  3801.8    .045       0
  4269.1     .07       0  4376.9    .045       0  4696.1     .07       0
    4946     .16       0  5026.9     .07       0  5044.1     .16       0
    5111     .07       0
Bank Sta=5026.9,5044.1
XS Rating Curve= 0 ,0
Exp/Cntr=0.3,0.1

Type RM Length L Ch R = 1 ,16500   ,500,500,500
BEGIN DESCRIPTION:
Stink Creek 32.0
END DESCRIPTION:
XS GIS Cut Line= 3
      1437005.01        6869588.      1439677.21      6870461.02
      1441554.99        6870388.
#Sta/Elev= 30
  2188.8 1971.17  2247.5 1970.83    2465 1968.38  2877.1 1953.52  3070.8    1946
  3235.4 1942.64  3272.6  1940.4  3282.9 1936.79  3291.5 1938.93  3407.6 1940.74
  3563.6 1941.34  3612.7 1941.81  4878.4 1942.13  4955.5 1941.49    4978 1936.96
  4978.6 1933.97  4979.1 1933.47  4995.8 1933.97  5017.8 1939.59    5075 1942.46
  5159.8 1941.21  5348.4  1943.5  5690.8 1950.36  5748.4 1953.58  5828.4 1953.52
  5849.1 1951.56  6008.7 1951.44  6388.8 1954.78  6814.5 1963.15  6879.2 1965.37
#Mann= 18 ,-1 , 0
  2188.8    .035       0  2247.5     .07       0  2877.1     .16       0
  3291.5     .07       0  3407.6    .045       0  3563.6     .07       0
  3612.7    .045       0  4878.4     .07       0  4955.5     .16       0
  4978.6     .07       0  4995.8     .16       0    5075     .07       0
  5159.8     .16       0  5348.4     .07       0  5690.8    .035       0
  5849.1     .07       0  6008.7     .05       0  6814.5     .07       0
#XS Ineff= 2 , 0
         4624.37 1951.91
Permanent Ineff=
       F       F
Bank Sta=4978.6,4995.8
XS Rating Curve= 0 ,0
Exp/Cntr=0.3,0.1

Type RM Length L Ch R = 1 ,16000   ,500,500,500
BEGIN DESCRIPTION:
Stink Creek 31.0
END DESCRIPTION:
XS GIS Cut Line= 3
      1437205.04      6869738.02      1439848.19      6870892.07
      1441754.99        6870388.
#Sta/Elev= 30
  2115.9 1970.09  2427.5  1960.7  2532.1 1961.87  2683.4 1951.72  2980.7 1946.84
  3049.7 1941.73    3156 1940.19  3202.3 1939.97  3239.8 1935.89  3261.6 1940.67
  3429.9 1940.86  4496.6 1940.59  4627.5 1941.04  4931.9 1939.32  4955.3 1936.81
  4970.1 1931.89  4970.6 1931.39  4987.4 1931.89  4995.5 1937.17  5017.4 1939.54
  5069.1 1938.08  5121.1  1940.6  5436.9  1944.4  5581.9 1946.34  5802.6 1948.27
  5856.2 1948.67  5903.5 1949.17  6013.8 1950.52  6669.2 1962.53  6972.3 1973.04
#Mann= 16 ,-1 , 0
  2115.9     .07       0  3049.7     .16       0    3156     .07       0
  3429.9    .045       0  4496.6     .07       0  4627.5     .16       0
  4970.1     .07       0  4987.4     .16       0  5121.1     .07       0
  5436.9    .035       0  5581.9     .05       0  5802.6     .07       0
  5856.2     .05       0  5903.5     .07       0  6013.8     .05       0
  6669.2     .07       0
Bank Sta=4970.1,4987.4
XS Rating Curve= 0 ,0
Exp/Cntr=0.3,0.1

Type RM Length L Ch R = 1 ,15500   ,403,403,403
BEGIN DESCRIPTION:
Stink Creek 30.0
END DESCRIPTION:
XS GIS Cut Line= 3
      1437555.03      6869938.02      1439573.02      6871170.71
      1441304.95        6871288.
#Sta/Elev= 30
  2635.3 1961.48  2693.9 1960.55    2765 1954.88    2854 1952.86  3070.8  1952.6
  3138.5 1944.16  3185.6 1942.36  3223.1 1941.39  3337.1  1939.1  3355.3 1938.92
  3370.7 1935.75  3376.6 1938.06  3430.6 1934.22    3456 1939.71  3603.8 1940.22
    4192 1939.02  4809.2 1937.05  4963.7 1936.44  4978.9 1935.25  4989.6 1929.88
  4990.1 1929.38  5006.9 1929.88  5030.5 1935.91  5071.1  1936.9  5593.7 1941.56
    5778 1943.06  6295.6 1949.23  6424.3 1951.63  6675.3 1956.97  6735.9 1957.62
#Mann= 16 ,-1 , 0
  2635.3     .07       0  3185.6     .16       0  3223.1     .07       0
  3337.1     .16       0  3430.6     .07       0  3603.8    .045       0
    4192     .07       0  4809.2     .16       0  4989.6     .07       0
  5006.9     .16       0  5071.1     .07       0  5593.7    .035       0
    5778     .05       0  6295.6     .07       0  6424.3     .05       0
  6675.3     .07       0
Bank Sta=4989.6,5006.9
XS Rating Curve= 0 ,0
Exp/Cntr=0.3,0.1

Type RM Length L Ch R = 1 ,15097   ,597,597,597
BEGIN DESCRIPTION:
Stink Creek 29.0
END DESCRIPTION:
XS GIS Cut Line= 3
       1437812.4      6870888.22      1439257.94      6871339.99
      1440905.04        6871338.
#Sta/Elev= 30
  3485.5 1951.22    3530 1950.02  3637.9 1951.06    3773 1948.51    3838 1944.58
  3849.3 1939.85  3865.2  1935.4  3896.8 1931.13  3902.9 1935.78  3931.5 1936.71
  4619.7 1934.55  4955.9 1935.82  4986.4 1935.71  4995.8 1933.47  4998.4 1928.03
  4998.9 1927.53  5015.7 1928.03  5017.1 1931.87  5027.1 1934.18  5037.1 1933.53
  5057.1 1936.14  5291.1 1937.53  5346.2 1937.61  5551.3 1938.16  5647.8 1938.74
  5710.3 1939.59  5876.1 1940.49  6085.2 1942.85  6554.7 1948.51  6647.1 1950.08
#Mann= 14 ,-1 , 0
  3485.5     .07       0  3849.3     .16       0  3931.5     .07       0
  4955.9     .16       0  4998.4     .07       0  5015.7     .16       0
  5291.1     .07       0  5346.2     .16       0  5551.3     .07       0
  5647.8     .16       0  5710.3     .07       0  5876.1    .035       0
  6085.2     .05       0  6554.7     .07       0
Bank Sta=4998.4,5015.7
XS Rating Curve= 0 ,0
Exp/Cntr=0.3,0.1

Type RM Length L Ch R = 1 ,14500   ,500,500,500
BEGIN DESCRIPTION:
Stink Creek 28.0
END DESCRIPTION:
XS GIS Cut Line= 3
      1437954.98      6871287.99      1439193.19      6871797.93
      1440385.89      6871705.18
#Sta/Elev= 30
  3660.9 1954.51  3693.4 1954.69  3769.1 1951.19  3841.2 1943.27  4050.3  1936.1
  4288.2 1933.59    4472 1933.64  4642.7 1930.85  4647.2 1928.32  4647.7 1927.82
  4664.5 1928.32  4677.5 1930.88  4688.3 1930.96  4701.4 1928.72  4744.2 1931.63
  4754.7 1930.88  4926.3 1933.94  4962.4 1928.99  4969.5  1930.9  4991.8 1930.88
  5002.3 1932.25  5106.7 1934.05  5803.1 1936.95  5844.4  1936.5  5884.5  1938.2
  5894.5 1937.25  5914.6 1938.76  6050.7  1941.7  6105.1 1944.35  6196.3 1945.02
#Mann= 9 ,-1 , 0
  3660.9     .07       0  3841.2     .16       0  4647.2     .07       0
  4664.5     .16       0  4744.2     .07       0  5002.3     .16       0
  5106.7     .07       0  5803.1    .035       0  6050.7     .05       0
Bank Sta=4647.2,4664.5
XS Rating Curve= 0 ,0
Exp/Cntr=0.3,0.1

Type RM Length L Ch R = 1 ,14000   ,1000,1000,1000
BEGIN DESCRIPTION:
Stink Creek 27.0
END DESCRIPTION:
XS GIS Cut Line= 5
        1438205.        6871538.      1438686.96      6871780.86
      1438925.03        6872088.      1439094.49      6872201.59
      1440350.27      6872159.27
#Sta/Elev= 30
  4071.7 1948.87  4102.4 1942.76  4124.7 1940.35  4201.1 1937.51  4316.8  1935.5
  4371.2 1934.91    4398 1935.03  4452.4 1931.59  4503.9 1933.24  4750.1 1930.26
  4772.3 1929.43  4779.1 1927.54  4814.4 1930.48  4928.4 1931.84  4963.8 1930.75
  4971.9 1929.44  4977.8 1925.48  4978.3 1924.98  4995.1 1925.48  4996.8 1928.23
  5028.5  1930.4  5094.5 1930.23  5100.5 1932.21  5115.5 1930.33  5121.5 1932.39
    5197 1932.75  6064.2 1933.79  6290.1 1936.25  6389.2 1938.02  6460.5 1940.83
#Mann= 10 ,-1 , 0
  4071.7     .07       0  4201.1     .16       0  4316.8     .07       0
  4371.2     .16       0  4977.8     .07       0  4995.1     .16       0
    5197     .07       0  6064.2    .035       0  6290.1     .07       0
  6389.2    .035       0
Bank Sta=4977.8,4995.1
XS Rating Curve= 0 ,0
Exp/Cntr=0.3,0.1

Type RM Length L Ch R = 1 ,13000   ,404,404,404
BEGIN DESCRIPTION:
Stink Creek 25.0
END DESCRIPTION:
XS GIS Cut Line= 4
      1437954.99      6871787.97      1438020.65      6871971.58
      1438410.96      6872242.43      1440400.86      6872443.46
#Sta/Elev= 30
    4805 1951.44  4879.9 1950.84  4938.2 1948.96  4953.7 1943.94    4969 1934.82
    4975  1929.1    4985 1923.81  4985.5 1923.31  5003.9 1923.81  5006.9 1925.67
  5021.8 1926.11  5087.3 1926.25    5138 1927.49  5190.2 1926.62  5382.5 1925.56
  5467.8 1926.59  5539.4 1928.92  5677.4 1930.62  6494.3 1931.82  6504.3 1932.53
  6877.4 1931.81  6966.7 1932.95  7005.8 1932.29  7107.4 1932.37  7161.6 1933.35
    7228 1933.01  7367.4 1936.13  7378.8 1935.57    7429 1936.25  7475.1 1938.85
#Mann= 7 ,-1 , 0
    4805     .07       0  4879.9     .16       0    4985     .07       0
  5003.9     .16       0  5190.2     .07       0  7005.8    .035       0
  7161.6     .07       0
Bank Sta=4985,5003.9
XS Rating Curve= 0 ,0
Exp/Cntr=0.3,0.1
