HEC-RAS study Sweetwater Creek.prj: Sweetwater Creek Base Level Engineering

--- Sweetwater Creek.g01 (geometry) --- (continued)

Type RM Length L Ch R = 1,319500,500,500,500
BEGIN DESCRIPTION:
Sweetwater Creek 637.0
END DESCRIPTION:
XS GIS Cut Line= 3
      1362905.03      6786387.98      1363381.93      6786115.01
      1364205.00      6785888.00
#Sta/Elev= 30
  4450.5 2487.17  4588.7 2480.41  4705.9 2478.06  4715.5 2477.63  4721.7 2475.89
  4743.3 2476.67  4750.1 2475.35  4830.7 2473.21  4947.7 2466.55  4992.0 2461.43
  4998.9 2462.72  5013.6 2461.40  5047.5 2463.22  5087.1 2466.74  5127.7 2466.34
  5148.4 2464.27  5155.8 2462.52  5157.8 2459.53  5158.3 2459.03  5180.5 2459.53
  5189.9 2464.28  5324.8 2466.96  5422.3 2472.04  5501.4 2484.52  5615.2 2492.44
  5667.1 2494.53  5723.2 2499.73  5802.3 2513.66  5822.7 2515.13  5853.8 2519.58
#Mann=3,-1,0
  4450.5    0.07       0  5157.8    0.07       0  5180.5    0.07       0
Bank Sta=5157.8,5180.5
Exp/Cntr=0.3,0.1

Type RM Length L Ch R = 1,319000,500,500,500
BEGIN DESCRIPTION:
Sweetwater Creek 636.0
END DESCRIPTION:
XS GIS Cut Line= 3
      1363054.98      6786688.01      1363404.92      6786575.46
      1364354.96      6786188.02
#Sta/Elev= 30
  4632.4 2485.92  4744.7 2477.24  4863.5 2472.12  4884.5 2474.12  4905.2 2469.29
  4979.9 2461.51  4986.1 2456.82  4986.6 2456.32  5008.8 2456.82  5011.4 2459.03
  5021.7 2460.59  5172.9 2466.50  5367.3 2463.12  5399.0 2459.45  5457.9 2461.18
  5496.9 2459.77  5506.0 2461.24  5535.4 2475.32  5588.9 2485.17  5637.0 2488.04
  5725.3 2485.84  5743.9 2488.59  5749.3 2486.55  5810.1 2490.96  5842.5 2490.69
  5896.5 2496.58  5928.4 2504.60  5933.8 2503.42  5987.3 2515.12  6026.0 2520.46
#Mann=3,-1,0
  4632.4    0.07       0  4986.1    0.07       0  5008.8    0.07       0
Bank Sta=4986.1,5008.8
Exp/Cntr=0.3,0.1

Type RM Length L Ch R = 1,318500,500,500,500
BEGIN DESCRIPTION:
Sweetwater Creek 635.0
END DESCRIPTION:
XS GIS Cut Line= 3
      1363204.98      6786988.01      1363682.48      6786864.16
      1364105.03      6786537.98
#Sta/Elev= 30
  4506.7 2485.33  4558.4 2483.36  4651.4 2475.79  4713.3 2474.60  4727.3 2472.04
  4767.9 2472.59  4878.6 2464.09  4889.6 2459.62  4919.9 2457.75  4925.0 2456.02
  4960.4 2457.49  4965.6 2456.03  4994.3 2454.92  4994.8 2454.42  5017.1 2454.92
  5028.4 2458.89  5041.1 2460.00  5113.5 2463.06  5198.6 2463.07  5213.1 2461.91
  5283.8 2463.49  5306.4 2461.61  5312.8 2458.77  5319.1 2458.00  5356.3 2458.88
  5362.6 2457.91  5397.9 2463.93  5426.9 2471.20  5433.2 2474.09  5533.8 2490.34
#Mann=3,-1,0
  4506.7    0.07       0  4994.3    0.07       0  5017.1    0.07       0
Bank Sta=4994.3,5017.1
Exp/Cntr=0.3,0.1

Type RM Length L Ch R = 1,318000,500,500,500
BEGIN DESCRIPTION:
Sweetwater Creek 634.0
END DESCRIPTION:
XS GIS Cut Line= 3
      1363354.96      6787338.01      1363706.60      6787245.52
      1364655.04      6786837.98
#Sta/Elev= 30
  4636.4 2482.12  4734.7 2474.40  4915.6 2468.03  4926.0 2466.84  4966.4 2455.22
  4993.6 2452.60  4994.1 2452.10  5016.4 2452.60  5063.6 2453.59  5081.1 2457.20
  5086.6 2455.42  5096.2 2456.24  5104.7 2459.14  5110.1 2456.39  5128.2 2459.95
  5133.7 2458.63  5238.8 2459.59  5338.4 2462.11  5409.0 2461.32  5432.6 2454.02
  5455.4 2454.56  5508.7 2465.72  5590.2 2473.58  5673.1 2490.27  5713.4 2494.62
  5818.5 2497.51  5934.3 2506.59  6010.5 2517.28  6017.8 2519.97  6032.3 2519.77
#Mann=3,-1,0
  4636.4    0.07       0  4993.6    0.07       0  5016.4    0.07       0
Bank Sta=4993.6,5016.4
Exp/Cntr=0.3,0.1

Type RM Length L Ch R = 1,317500,500,500,500
BEGIN DESCRIPTION:
Sweetwater Creek 633.0
END DESCRIPTION:
XS GIS Cut Line= 3
      1363755.01      6788037.98      1363954.35      6787650.89
      1364354.98      6787138.02
#Sta/Elev= 30
  4564.6 2475.17  4632.1 2474.25  4677.1 2471.01  4705.9 2466.37  4728.0 2469.12
  4744.5 2466.85  4750.2 2464.38  4755.8 2460.02  4772.4 2458.13  4855.4 2457.19
  4944.1 2451.95  4951.2 2450.51  4951.7 2450.01  4981.4 2450.51  5004.6 2452.04
  5009.6 2454.41  5030.4 2456.93  5059.3 2458.31  5138.0 2458.34  5158.8 2459.87
  5202.2 2459.37  5272.8 2461.19  5295.4 2460.37  5301.7 2461.39  5314.8 2458.11
  5325.5 2458.85  5337.0 2462.27  5459.1 2464.96  5558.6 2470.61  5650.8 2483.02
#Mann=5,-1,0
  4564.6    0.07       0  4951.2    0.07       0  4981.4    0.07       0
  5314.8    0.16       0  5325.5    0.07       0
Bank Sta=4951.2,4981.4
Exp/Cntr=0.3,0.1

Type RM Length L Ch R = 1,317000,500,500,500
BEGIN DESCRIPTION:
Sweetwater Creek 632.0
END DESCRIPTION:
XS GIS Cut Line= 3
      1364104.99      6788238.03      1364174.90      6788007.39
      1364554.98      6787638.01
#Sta/Elev= 30
  4759.0 2471.59  4769.5 2472.10  4775.5 2471.05  4832.2 2470.36  4874.0 2468.14
  4884.7 2466.68  4926.2 2464.09  4936.7 2462.98  4950.5 2460.49  4968.0 2450.12
  4978.2 2448.99  4988.9 2448.75  4991.6 2447.94  4992.1 2447.44  5021.3 2447.44
  5021.8 2447.94  5028.0 2452.21  5042.0 2454.88  5056.1 2455.04  5084.4 2454.03
  5183.4 2457.48  5233.0 2457.94  5254.2 2458.94  5346.2 2460.56  5452.2 2464.93
  5494.7 2467.35  5508.8 2468.79  5522.9 2469.48  5526.5 2470.75  5530.0 2470.75
#Mann=3,-1,0
  4759.0    0.07       0  4991.6    0.07       0  5021.8    0.07       0
Bank Sta=4991.6,5021.8
Exp/Cntr=0.3,0.1

Type RM Length L Ch R = 1,316500,500,500,500
BEGIN DESCRIPTION:
Sweetwater Creek 631.0
END DESCRIPTION:
XS GIS Cut Line= 3
      1364155.01      6788438.00      1364508.00      6788333.27
      1364904.97      6787988.02
#Sta/Elev= 30
  4631.8 2470.67  4653.6 2469.28  4663.1 2467.50  4673.5 2467.92  4686.8 2466.42
  4704.8 2469.15  4720.1 2468.28  4725.7 2466.80  4819.5 2464.45  4913.4 2460.61
  4935.1 2458.53  4976.0 2448.52  5007.4 2447.18  5007.9 2446.68  5037.7 2447.18
  5050.9 2452.54  5072.8 2453.18  5101.2 2452.20  5207.6 2455.45  5313.9 2455.93
  5355.7 2458.71  5369.9 2462.17  5377.5 2466.49  5384.2 2468.11  5412.7 2482.32
  5420.1 2488.89  5426.9 2491.41  5441.2 2494.22  5469.6 2497.25  5526.1 2500.26
#Mann=3,-1,0
  4631.8    0.07       0  5007.4    0.07       0  5037.7    0.07       0
Bank Sta=5007.4,5037.7
Exp/Cntr=0.3,0.1

Type RM Length L Ch R = 1,316000,500,500,500
BEGIN DESCRIPTION:
Sweetwater Creek 630.0
END DESCRIPTION:
XS GIS Cut Line= 3
      1364355.03      6789037.98      1364857.63      6788640.31
      1365104.96      6788588.01
#Sta/Elev= 30
  4359.1 2465.45  4550.6 2461.71  4565.0 2461.05  4587.5 2458.13  4593.9 2458.09
  4608.3 2462.62  4614.7 2462.87  4643.5 2458.74  4658.0 2459.63  4779.8 2456.59
  4786.2 2455.73  4881.7 2452.26  4949.7 2445.93  4964.1 2446.66  4969.8 2444.35
  4970.3 2443.85  5000.1 2444.35  5008.5 2447.37  5039.3 2450.84  5089.3 2449.65
  5109.7 2451.11  5120.0 2454.82  5128.5 2459.53  5133.6 2460.70  5140.4 2465.08
  5150.6 2479.73  5160.8 2491.65  5171.1 2495.70  5191.5 2497.05  5252.8 2498.72
#Mann=5,-1,0
  4359.1    0.07       0  4881.7    0.16       0  4969.8    0.07       0
  5000.1    0.16       0  5008.5    0.07       0
Bank Sta=4969.8,5000.1
Exp/Cntr=0.3,0.1

Type RM Length L Ch R = 1,315500,500,500,500
BEGIN DESCRIPTION:
Sweetwater Creek 629.0
END DESCRIPTION:
XS GIS Cut Line= 3
      1364854.99      6789438.01      1365054.62      6789050.17
      1365155.02      6788987.99
#Sta/Elev= 30
  4563.8 2477.01  4572.1 2477.19  4577.7 2474.43  4594.3 2470.98  4599.9 2468.34
  4631.3 2459.00  4644.2 2452.60  4660.8 2452.27  4666.4 2455.27  4683.0 2459.07
  4698.8 2455.79  4710.7 2450.84  4727.3 2447.94  4749.5 2451.06  4838.2 2449.78
  4904.7 2445.30  4921.2 2446.81  4943.4 2446.70  4965.6 2444.35  4971.2 2442.52
  4980.0 2442.52  4987.7 2444.24  4993.4 2442.92  5003.2 2443.13  5008.8 2441.01
  5009.3 2440.51  5039.2 2441.01  5073.8 2455.06  5095.0 2460.20  5118.1 2463.68
#Mann=3,-1,0
  4563.8    0.07       0  5008.8    0.07       0  5039.2    0.07       0
Bank Sta=5008.8,5039.2
Exp/Cntr=0.3,0.1

Type RM Length L Ch R = 1,315000,500,500,500
BEGIN DESCRIPTION:
Sweetwater Creek 628.0
END DESCRIPTION:
XS GIS Cut Line= 3
      1365005.04      6789537.98      1365211.50      6789444.34
      1365454.98      6788938.04
#Sta/Elev= 30
  4773.3 2465.00  4776.0 2465.00  4805.1 2456.11  4828.2 2459.31  4849.5 2451.60
  4862.3 2445.52  4872.1 2444.22  4879.9 2444.73  4894.0 2448.35  4938.0 2447.90
  4948.9 2446.58  4954.6 2443.96  4955.6 2439.80  4956.1 2439.30  4986.2 2439.80
  4992.9 2441.35  5007.0 2441.44  5045.2 2444.40  5061.4 2445.03  5066.9 2443.73
  5095.8 2445.98  5106.6 2445.49  5157.4 2447.28  5185.6 2450.38  5276.2 2456.70
  5338.5 2459.73  5395.4 2466.08  5457.2 2469.91  5508.0 2477.35  5561.8 2482.65
#Mann=5,-1,0
  4773.3    0.07       0  4849.5    0.16       0  4955.6    0.07       0
  4986.2    0.16       0  5045.2    0.07       0
Bank Sta=4955.6,4986.2
Exp/Cntr=0.3,0.1

Type RM Length L Ch R = 1,314500,500,500,500
BEGIN DESCRIPTION:
Sweetwater Creek 627.0
END DESCRIPTION:
XS GIS Cut Line= 3
      1365505.01      6790037.96      1365558.67      6789779.67
      1365655.00      6789288.02
#Sta/Elev= 30
  4736.2 2468.47  4756.1 2466.90  4777.0 2464.04  4787.2 2460.46  4797.4 2454.58
  4806.2 2447.32  4811.3 2444.42  4817.9 2443.07  4838.3 2443.99  4888.0 2442.76
  4899.6 2443.51  4920.0 2442.37  4950.6 2439.19  4961.7 2436.77  4971.1 2439.43
  5003.4 2441.13  5006.8 2436.08  5007.3 2435.58  5037.4 2436.08  5042.5 2440.33
  5049.6 2441.67  5063.4 2445.80  5073.0 2447.68  5114.9 2447.86  5144.4 2449.23
  5174.9 2449.17  5269.4 2451.93  5315.7 2454.28  5367.2 2455.82  5501.0 2463.63
#Mann=5,-1,0
  4736.2    0.07       0  4888.0    0.16       0  5006.8    0.07       0
  5037.4    0.16       0  5049.6    0.07       0
Bank Sta=5006.8,5037.4
Exp/Cntr=0.3,0.1

Type RM Length L Ch R = 1,314000,500,500,500
BEGIN DESCRIPTION:
Sweetwater Creek 626.0
END DESCRIPTION:
XS GIS Cut Line= 3
      1365654.99      6790188.00      1365876.51      6790108.66
      1366105.01      6789587.99
#Sta/Elev= 30
  4764.7 2468.96  4796.6 2468.05  4836.3 2463.86  4841.6 2464.44  4860.3 2461.19
  4872.4 2460.97  4881.6 2458.50  4913.4 2454.88  4923.3 2451.98  4928.6 2447.79
  4945.3 2438.98  4954.0 2435.42  4961.8 2433.47  4962.3 2432.97  4992.5 2433.47
  4996.5 2437.02  5003.1 2437.02  5012.9 2438.79  5044.4 2438.50  5059.6 2439.18
  5077.2 2442.69  5083.0 2443.03  5153.1 2444.49  5175.4 2445.77  5317.4 2445.17
  5372.0 2446.02  5426.4 2448.55  5478.6 2454.14  5536.3 2457.69  5568.6 2458.74
#Mann=3,-1,0
  4764.7    0.07       0  4961.8    0.07       0  4992.5    0.07       0
Bank Sta=4961.8,4992.5
Exp/Cntr=0.3,0.1

Type RM Length L Ch R = 1,313500,500,500,500
BEGIN DESCRIPTION:
Sweetwater Creek 625.0
END DESCRIPTION:
XS GIS Cut Line= 3
      1366055.00      6790487.99      1366271.69      6790237.64
      1366654.98      6789888.02
#Sta/Elev= 30
  4668.9 2454.64  4704.5 2453.81  4782.4 2445.92  4888.8 2443.05  4895.4 2442.48
  4903.0 2440.13  4909.7 2439.80  4917.3 2437.78  4959.9 2434.96  4993.7 2431.45
  4994.2 2430.95  5024.4 2431.45  5037.4 2436.32  5058.6 2440.15  5072.6 2440.44
  5080.0 2439.56  5094.2 2435.97  5115.1 2437.50  5136.8 2437.52  5165.1 2440.18
  5203.5 2439.91  5228.6 2439.71  5285.6 2444.72  5328.0 2451.13  5356.3 2453.15
  5405.7 2461.54  5483.4 2468.18  5511.7 2472.82  5515.4 2475.01  5518.8 2475.01
#Mann=5,-1,0
  4668.9    0.07       0  4993.7    0.07       0  5024.4    0.07       0
  5203.5    0.16       0  5285.6    0.07       0
Bank Sta=4993.7,5024.4
Exp/Cntr=0.3,0.1

Type RM Length L Ch R = 1,313000,500,500,500
BEGIN DESCRIPTION:
Sweetwater Creek 624.0
END DESCRIPTION:
XS GIS Cut Line= 3
      1365705.00      6790588.00      1366691.00      6790401.36
      1366804.98      6790338.01
#Sta/Elev= 30
  3996.5 2459.23  4237.1 2455.23  4393.4 2454.16  4434.1 2451.91  4515.6 2444.30
  4769.7 2441.79  4820.9 2440.42  4841.2 2436.76  4861.6 2435.76  4885.3 2437.09
  4937.4 2435.06  4943.0 2431.67  4963.4 2432.57  4973.5 2430.98  4983.7 2428.27
  4983.9 2427.35  4984.4 2426.85  5015.1 2427.35  5022.6 2445.99  5027.5 2458.22
  5035.5 2465.83  5041.2 2463.37  5050.3 2469.96  5057.2 2477.39  5073.2 2484.16
  5079.0 2489.78  5084.7 2490.18  5095.0 2494.36  5107.5 2496.86  5130.4 2497.62
#Mann=6,-1,0
  3996.5    0.07       0  4769.7    0.16       0  4937.4    0.07       0
  4983.9    0.07       0  5015.1    0.07       0  5022.6    0.07       0
Bank Sta=4983.9,5015.1
Exp/Cntr=0.3,0.1

Type RM Length L Ch R = 1,312500,500,500,500
BEGIN DESCRIPTION:
Sweetwater Creek 623.0
END DESCRIPTION:
XS GIS Cut Line= 3
      1366254.96      6790687.98      1366604.47      6790872.87
      1366704.99      6790838.00
#Sta/Elev= 30
  4604.6 2450.93  4649.9 2448.70  4678.8 2445.92  4684.5 2446.01  4700.8 2443.99
  4722.9 2443.24  4739.2 2441.28  4761.2 2439.96  4810.9 2438.98  4849.2 2439.46
  4898.9 2438.29  4915.2 2436.42  4921.4 2434.28  4931.6 2432.48  4975.6 2428.64
  4981.3 2428.87  4995.6 2426.65  4996.1 2426.15  5026.3 2426.15  5026.8 2426.65
  5028.6 2435.02  5033.9 2432.96  5042.9 2441.40  5053.5 2455.16  5059.7 2468.79
  5065.0 2469.04  5074.7 2476.11  5085.2 2479.50  5090.8 2481.98  5106.4 2484.01
#Mann=3,-1,0
  4604.6    0.07       0  4995.6    0.07       0  5026.8    0.07       0
Bank Sta=4995.6,5026.8
Exp/Cntr=0.3,0.1

Type RM Length L Ch R = 1,312000,500,500,500
BEGIN DESCRIPTION:
Sweetwater Creek 622.0
END DESCRIPTION:
XS GIS Cut Line= 3
      1365640.51      6790768.48      1366454.21      6791324.80
      1366640.81      6791173.71
#Sta/Elev= 30
  4014.3 2462.37  4014.6 2462.37  4031.9 2460.43  4039.0 2456.56  4074.9 2452.34
  4189.3 2446.64  4241.8 2447.64  4377.9 2444.74  4592.2 2437.98  4616.1 2439.18
  4693.8 2437.87  4735.8 2431.60  4744.6 2436.14  4758.7 2436.49  4849.0 2434.16
  4930.1 2430.86  4952.5 2428.15  4960.0 2425.22  4980.9 2426.87  4982.8 2424.51
  4983.3 2424.01  5014.0 2424.51  5019.5 2424.93  5033.9 2436.20  5040.4 2434.55
  5048.3 2440.83  5054.7 2440.45  5062.7 2445.02  5118.7 2446.71  5240.1 2461.84
#Mann=8,-1,0
  4014.3   0.035       0  4014.6    0.07       0  4241.8    0.16       0
  4377.9    0.07       0  4616.1    0.16       0  4849.0    0.07       0
  4982.8    0.07       0  5014.0    0.07       0
Bank Sta=4982.8,5014
Exp/Cntr=0.3,0.1

Type RM Length L Ch R = 1,311500,500,500,500
BEGIN DESCRIPTION:
Sweetwater Creek 621.0
END DESCRIPTION:
XS GIS Cut Line= 3
      1365854.96      6791838.01      1366204.07      6791725.46
      1366557.66      6791520.30
#Sta/Elev= 30
  4633.2 2482.86  4686.6 2479.18  4700.2 2475.48  4706.8 2472.98  4713.4 2465.84
  4718.6 2463.36  4745.4 2462.51  4777.5 2441.96  4809.5 2432.23  4814.8 2433.74
  4841.6 2428.07  4948.4 2429.19  4959.0 2428.51  4975.1 2424.03  4980.3 2424.66
  4990.1 2423.00  4990.6 2422.50  5021.7 2423.00  5027.4 2425.79  5070.4 2425.45
  5101.9 2428.50  5107.7 2427.27  5123.5 2429.51  5197.6 2431.36  5219.5 2433.78
  5225.3 2433.06  5241.0 2435.83  5246.8 2434.26  5262.6 2436.34  5408.8 2437.15
#Mann=4,-1,0
  4633.2   0.035       0  4700.2    0.07       0  4990.1    0.07       0
  5021.7    0.07       0
Bank Sta=4990.1,5021.7
Exp/Cntr=0.3,0.1

Type RM Length L Ch R = 1,311000,500,500,500
BEGIN DESCRIPTION:
Sweetwater Creek 620.0
END DESCRIPTION:
XS GIS Cut Line= 3
      1366254.98      6792238.04      1366298.42      6792131.77
      1366804.98      6791138.04
#Sta/Elev= 30
  4885.2 2450.15  4900.0 2450.37  4917.7 2448.50  4924.0 2446.41  4929.4 2443.20
  4937.6 2420.21  4938.1 2419.71  4969.2 2420.21  4971.7 2421.07  5015.5 2421.48
  5037.9 2423.81  5051.1 2423.91  5105.3 2429.72  5140.1 2431.95  5318.5 2436.36
  5401.3 2437.05  5543.0 2434.17  5700.1 2437.87  5757.0 2438.20  5818.1 2439.18
  5834.7 2438.54  5865.4 2440.94  5884.8 2441.82  5907.0 2445.31  5923.6 2450.50
  5929.3 2450.72  5980.8 2460.76  6018.2 2463.63  6048.1 2467.48  6115.4 2468.43
#Mann=5,-1,0
  4885.2    0.07       0  4937.6    0.07       0  4969.2    0.07       0
  5757.0    0.16       0  5865.4    0.07       0
Bank Sta=4937.6,4969.2
Exp/Cntr=0.3,0.1

Type RM Length L Ch R = 1,310500,500,500,500
BEGIN DESCRIPTION:
Sweetwater Creek 619.0
END DESCRIPTION:
XS GIS Cut Line= 3
      1366804.99      6792087.99      1366708.98      6791984.45
      1366505.00      6791788.00
#Sta/Elev= 30
  4858.8 2447.79  4865.9 2448.37  4908.4 2449.19  4915.2 2448.53  4922.6 2447.07
  4929.4 2436.99  4936.7 2427.72  4943.5 2422.87  4950.9 2421.28  4957.7 2418.51
  4963.4 2414.77  4963.9 2414.27  4994.6 2414.27  4995.1 2414.77  4999.3 2417.00
  5007.3 2417.82  5021.4 2420.50  5028.6 2422.40  5042.8 2423.43  5063.9 2426.35
  5071.1 2428.44  5078.0 2428.34  5085.2 2429.84  5106.3 2431.54  5113.5 2432.60
  5148.8 2434.75  5156.0 2434.70  5162.9 2435.45  5191.2 2436.39  5283.2 2437.00
#Mann=3,-1,0
  4858.8    0.07       0  4963.4    0.07       0  4995.1    0.07       0
Bank Sta=4963.4,4995.1
Exp/Cntr=0.3,0.1

Type RM Length L Ch R = 1,310000,500,500,500
BEGIN DESCRIPTION:
Sweetwater Creek 618.0
END DESCRIPTION:
XS GIS Cut Line= 3
      1366955.01      6791938.04      1366851.69      6791532.70
      1366805.00      6791338.02
#Sta/Elev= 30
  4581.7 2435.46  4612.7 2435.53  4645.6 2434.23  4654.0 2433.17  4674.6 2432.90
  4736.5 2426.31  4792.7 2424.06  4829.4 2423.65  4844.9 2424.41  4870.7 2422.87
  4880.6 2423.30  4885.8 2422.37  4912.0 2422.14  4942.9 2420.66  4953.3 2418.71
  4973.9 2418.58  4984.0 2411.43  4984.5 2410.93  5015.7 2411.43  5025.4 2416.49
  5045.5 2420.91  5050.6 2423.75  5056.2 2425.35  5087.1 2424.49  5097.8 2431.49
  5134.6 2437.57  5148.8 2441.08  5159.1 2441.60  5173.4 2443.89  5200.2 2448.14
#Mann=5,-1,0
  4581.7    0.07       0  4792.7    0.16       0  4984.0    0.07       0
  5015.7    0.16       0  5173.4    0.07       0
Bank Sta=4984,5015.7
Exp/Cntr=0.3,0.1

Type RM Length L Ch R = 1,309500,500,500,500
BEGIN DESCRIPTION:
Sweetwater Creek 617.0
END DESCRIPTION:
XS GIS Cut Line= 3
      1367055.02      6791887.97      1367235.26      6791618.37
      1367355.00      6791438.00
#Sta/Elev= 30
  4675.7 2434.11  4761.3 2431.11  4832.8 2429.82  4869.4 2427.50  4920.4 2421.33
  4935.4 2421.61  4941.4 2419.20  4956.5 2414.88  4970.6 2411.94  4971.1 2411.44
  5001.9 2411.44  5002.4 2411.94  5003.2 2413.34  5007.5 2414.17  5022.6 2414.37
  5049.6 2416.20  5058.6 2417.69  5064.6 2420.12  5072.5 2425.31  5079.7 2432.86
  5085.7 2441.48  5094.7 2462.12  5100.7 2472.49  5108.5 2477.93  5115.8 2480.52
  5136.8 2480.28  5151.9 2478.25  5157.9 2479.68  5166.9 2479.13  5216.5 2481.55
#Mann=4,-1,0
  4675.7    0.07       0  4832.8    0.16       0  4970.6    0.07       0
  5002.4    0.16       0
Bank Sta=4970.6,5002.4
Exp/Cntr=0.3,0.1

Type RM Length L Ch R = 1,309000,500,500,500
BEGIN DESCRIPTION:
Sweetwater Creek 616.0
END DESCRIPTION:
XS GIS Cut Line= 3
      1367105.02      6791938.00      1367441.12      6792001.24
      1367555.03      6791937.98
#Sta/Elev= 30
  4658.0 2433.63  4684.2 2431.58  4719.0 2430.19  4786.1 2429.13  4841.1 2428.10
  4851.8 2427.34  4871.7 2422.92  4892.0 2420.68  4899.2 2418.81  4904.3 2419.13
  4907.3 2418.40  4912.4 2417.15  4932.7 2415.20  4983.6 2413.12  5003.4 2410.23
  5003.9 2409.73  5034.7 2409.73  5035.2 2410.23  5035.3 2410.75  5041.0 2411.35
  5050.2 2410.75  5057.0 2413.17  5078.8 2417.48  5084.5 2421.70  5100.5 2428.31
  5107.4 2448.86  5116.5 2469.81  5122.3 2472.93  5127.4 2479.62  5130.3 2479.62
#Mann=5,-1,0
  4658.0    0.07       0  4786.1    0.16       0  4907.3    0.07       0
  5003.4    0.07       0  5035.2    0.07       0
Bank Sta=5003.4,5035.2
Exp/Cntr=0.3,0.1

Type RM Length L Ch R = 1,308500,500,500,500
BEGIN DESCRIPTION:
Sweetwater Creek 615.0
END DESCRIPTION:
XS GIS Cut Line= 3
      1366855.02      6792138.01      1367354.64      6792472.59
      1367455.04      6792437.99
#Sta/Elev= 30
  4398.7 2445.17  4463.2 2441.62  4493.2 2436.98  4499.2 2437.02  4550.3 2431.08
  4751.4 2425.54  4802.6 2420.86  4853.5 2418.95  4868.0 2416.02  4874.5 2413.20
  4880.5 2412.62  4889.5 2414.26  4895.5 2412.71  4916.5 2412.80  4946.5 2409.67
  4976.4 2409.55  4988.6 2408.76  4995.1 2407.51  4995.6 2407.01  5026.9 2407.51
  5028.1 2415.96  5033.4 2414.36  5053.3 2426.46  5059.3 2431.83  5064.6 2430.77
  5085.0 2457.71  5090.5 2463.12  5095.8 2463.24  5103.5 2468.99  5106.2 2468.99
#Mann=4,-1,0
  4398.7    0.07       0  4802.6    0.16       0  4995.1    0.07       0
  5026.9    0.16       0
Bank Sta=4995.1,5026.9
Exp/Cntr=0.3,0.1

Type RM Length L Ch R = 1,308000,500,500,500
BEGIN DESCRIPTION:
Sweetwater Creek 614.0
END DESCRIPTION:
XS GIS Cut Line= 3
      1366954.97      6792837.99      1367155.00      6792893.92
      1367555.01      6792838.00
#Sta/Elev= 30
  4792.3 2426.19  4802.7 2425.41  4809.4 2423.22  4833.9 2418.38  4865.0 2416.81
  4875.4 2417.66  4896.2 2416.62  4922.2 2412.04  4927.4 2414.37  4948.1 2408.87
  4979.2 2406.39  4982.4 2404.72  4982.9 2404.22  5014.2 2404.72  5020.2 2407.12
  5040.4 2410.79  5080.3 2411.93  5131.3 2410.52  5171.7 2413.21  5191.9 2418.69
  5220.2 2424.64  5225.3 2423.30  5232.2 2425.10  5282.7 2432.95  5291.7 2435.21
  5296.7 2435.43  5314.0 2441.95  5353.4 2449.88  5383.7 2453.89  5403.9 2453.35
#Mann=5,-1,0
  4792.3    0.07       0  4982.4    0.07       0  5014.2    0.07       0
  5080.3    0.16       0  5314.0    0.07       0
Bank Sta=4982.4,5014.2
Exp/Cntr=0.3,0.1

Type RM Length L Ch R = 1,307500,500,500,500
BEGIN DESCRIPTION:
Sweetwater Creek 613.0
END DESCRIPTION:
XS GIS Cut Line= 3
      1366955.00      6793488.00      1367162.18      6793392.58
      1367555.03      6792887.97
#Sta/Elev= 30
  4771.9 2443.41  4803.6 2442.01  4809.1 2440.57  4855.0 2445.31  4860.5 2440.09
  4871.0 2437.75  4883.5 2415.03  4893.0 2411.55  4915.0 2408.11  4952.4 2408.68
  4981.1 2407.01  4982.2 2403.15  4982.7 2402.65  5014.3 2403.15  5126.4 2407.44
  5147.2 2404.59  5155.4 2405.47  5176.2 2410.57  5219.6 2412.73  5226.0 2415.04
  5240.4 2414.46  5246.8 2416.78  5261.3 2417.92  5482.9 2426.24  5532.7 2431.04
  5556.1 2434.78  5567.1 2436.98  5611.4 2445.18  5632.2 2445.96  5639.5 2447.50
#Mann=5,-1,0
  4771.9    0.07       0  4982.2    0.07       0  5014.3    0.07       0
  5556.1    0.16       0  5567.1    0.07       0
Bank Sta=4982.2,5014.3
Exp/Cntr=0.3,0.1

Type RM Length L Ch R = 1,307000,500,500,500
BEGIN DESCRIPTION:
Sweetwater Creek 612.0
END DESCRIPTION:
XS GIS Cut Line= 3
      1367454.98      6793788.04      1367501.62      6793681.94
      1367904.99      6793188.02
#Sta/Elev= 30
  4884.1 2434.44  4916.4 2435.06  4960.6 2433.06  4968.6 2408.04  4982.5 2402.27
  4999.4 2400.09  5002.8 2397.95  5003.3 2397.45  5034.9 2397.95  5043.1 2400.74
  5061.9 2403.31  5082.7 2403.44  5125.8 2406.44  5146.8 2411.60  5168.9 2412.03
  5175.4 2409.94  5189.7 2410.47  5197.6 2412.44  5305.2 2417.13  5353.7 2419.50
  5428.9 2419.87  5488.4 2420.75  5537.9 2426.98  5545.8 2429.52  5552.3 2430.05
  5566.6 2434.84  5601.8 2450.27  5624.1 2457.37  5634.5 2462.48  5637.7 2462.48
#Mann=7,-1,0
  4884.1    0.07       0  5002.8    0.07       0  5034.9    0.07       0
  5043.1   0.035       0  5146.8    0.16       0  5305.2    0.07       0
  5428.9    0.16       0
Bank Sta=5002.8,5034.9
Exp/Cntr=0.3,0.1

Type RM Length L Ch R = 1,306500,500,500,500
BEGIN DESCRIPTION:
Sweetwater Creek 611.0
END DESCRIPTION:
XS GIS Cut Line= 3
      1367905.00      6794088.01      1367947.89      6793840.50
      1368354.99      6793488.00
#Sta/Elev= 30
  4748.8 2418.92  4850.3 2418.57  4901.0 2407.20  4955.3 2403.04  4956.0 2395.30
  4956.5 2394.80  4988.1 2395.30  4988.3 2395.39  4992.4 2397.15  5028.0 2398.67
  5049.1 2401.30  5113.5 2399.69  5127.8 2400.25  5134.4 2402.76  5139.3 2403.10
  5155.2 2407.68  5181.3 2407.79  5283.5 2406.82  5312.0 2407.78  5326.3 2409.97
  5340.1 2413.57  5368.0 2418.23  5389.9 2424.92  5418.4 2438.16  5432.6 2447.50
  5449.8 2457.00  5460.1 2463.09  5474.4 2466.13  5517.1 2467.48  5538.5 2466.79
#Mann=7,-1,0
  4748.8    0.07       0  4956.0    0.07       0  4988.1    0.07       0
  4988.3    0.16       0  5139.3    0.07       0  5181.3    0.16       0
  5449.8    0.07       0
Bank Sta=4956,4988.1
Exp/Cntr=0.3,0.1

Type RM Length L Ch R = 1,306000,500,500,500
BEGIN DESCRIPTION:
Sweetwater Creek 610.0
END DESCRIPTION:
XS GIS Cut Line= 3
      1368055.00      6794088.00      1368401.62      6793981.57
      1368504.98      6793788.04
#Sta/Elev= 30
  4637.4 2417.47  4659.0 2415.03  4668.8 2411.64  4700.2 2406.53  4757.2 2405.84
  4773.4 2405.05  4795.1 2401.25  4821.9 2401.65  4860.6 2403.15  4951.2 2400.69
  4972.1 2397.79  4991.5 2397.02  4996.7 2395.28  4997.6 2392.96  4998.2 2392.46
  5029.8 2392.96  5035.7 2394.69  5049.4 2395.52  5079.6 2403.95  5129.2 2411.64
  5145.5 2417.20  5151.4 2420.97  5161.7 2425.08  5174.1 2432.35  5183.7 2435.30
  5189.4 2439.92  5196.8 2443.71  5205.6 2445.71  5209.1 2445.50  5219.4 2446.01
#Mann=5,-1,0
  4637.4    0.07       0  4821.9    0.16       0  4997.6    0.07       0
  5029.8    0.16       0  5209.1    0.07       0
Bank Sta=4997.6,5029.8
Exp/Cntr=0.3,0.1

Type RM Length L Ch R = 1,305500,500,500,500
BEGIN DESCRIPTION:
Sweetwater Creek 609.0
END DESCRIPTION:
XS GIS Cut Line= 3
      1368004.98      6794238.00      1368525.29      6794288.00
      1368754.97      6794387.98
#Sta/Elev= 30
  4477.3 2417.82  4587.8 2417.12  4633.6 2413.96  4678.2 2412.51  4833.9 2409.66
  4838.6 2409.10  4843.6 2410.00  4889.2 2399.17  4919.3 2395.98  4929.4 2397.17
  4939.2 2395.10  4951.1 2393.94  4979.6 2396.40  4989.7 2394.80  4997.3 2391.20
  5002.6 2391.20  5003.6 2387.66  5004.4 2387.16  5039.5 2387.66  5043.3 2391.99
  5084.6 2393.10  5113.5 2396.40  5130.6 2413.14  5136.9 2428.38  5142.4 2430.80
  5152.4 2433.03  5174.2 2434.55  5206.9 2434.69  5241.5 2434.18  5250.5 2432.79
#Mann=5,-1,0
  4477.3    0.07       0  4833.9    0.16       0  4939.2    0.07       0
  5003.6    0.07       0  5039.5    0.07       0
Bank Sta=5003.6,5039.5
Exp/Cntr=0.3,0.1

Type RM Length L Ch R = 1,305000,500,500,500
BEGIN DESCRIPTION:
Sweetwater Creek 608.0
END DESCRIPTION:
XS GIS Cut Line= 3
      1368104.99      6794688.00      1368454.95      6794751.07
      1368705.02      6794687.99
#Sta/Elev= 30
  4644.4 2411.11  4664.7 2409.66  4676.3 2407.21  4685.1 2406.68  4847.6 2404.71
  4878.1 2401.19  4908.6 2399.76  4939.1 2391.59  4949.2 2390.89  4954.4 2388.12
  4959.5 2389.02  4969.6 2386.86  4971.9 2384.97  4972.7 2384.47  5007.8 2384.97
  5010.4 2388.37  5029.4 2391.90  5034.6 2391.58  5041.3 2392.90  5061.9 2392.88
  5075.6 2391.57  5111.6 2390.62  5116.7 2392.21  5152.6 2391.55  5157.8 2392.56
  5175.4 2392.94  5198.9 2395.95  5239.9 2405.97  5247.6 2407.41  5257.9 2408.09
#Mann=3,-1,0
  4644.4    0.07       0  4971.9    0.07       0  5007.8    0.16       0
Bank Sta=4971.9,5007.8
Exp/Cntr=0.3,0.1

Type RM Length L Ch R = 1,304500,500,500,500
BEGIN DESCRIPTION:
Sweetwater Creek 607.0
END DESCRIPTION:
XS GIS Cut Line= 3
      1368305.00      6795388.00      1368655.46      6795147.58
      1368905.05      6795087.99
#Sta/Elev= 30
  4575.0 2435.69  4598.6 2436.09  4660.2 2436.03  4696.3 2434.31  4705.0 2430.66
  4711.0 2419.96  4719.9 2413.15  4725.9 2409.79  4732.6 2403.16  4746.9 2396.00
  4761.8 2390.54  4776.7 2389.13  4823.9 2391.96  4890.4 2392.64  4914.1 2391.64
  4920.2 2392.44  4935.1 2386.50  4941.1 2388.21  4950.0 2386.00  4956.0 2387.13
  4963.1 2384.80  4970.9 2384.10  4996.7 2384.37  4999.3 2382.22  5000.2 2381.72
  5035.3 2382.22  5040.6 2390.86  5050.9 2397.36  5126.5 2401.16  5256.6 2405.34
#Mann=6,-1,0
  4575.0   0.035       0  4598.6    0.07       0  4823.9    0.16       0
  4999.3    0.07       0  5035.3    0.16       0  5126.5    0.07       0
Bank Sta=4999.3,5035.3
Exp/Cntr=0.3,0.1

Type RM Length L Ch R = 1,304000,500,500,500
BEGIN DESCRIPTION:
Sweetwater Creek 606.0
END DESCRIPTION:
XS GIS Cut Line= 3
      1368204.97      6795387.98      1368563.05      6795584.15
      1369854.99      6795688.00
#Sta/Elev= 30
  4591.7 2436.43  4681.3 2433.36  4831.4 2421.76  4873.7 2413.83  4893.7 2408.23
  4959.1 2398.78  4975.3 2393.19  4982.3 2396.09  4990.8 2394.49  4997.1 2387.20
  5003.5 2388.54  5004.0 2378.56  5004.9 2378.06  5040.0 2378.56  5042.1 2382.93
  5072.2 2389.31  5142.4 2388.58  5229.0 2392.19  5373.1 2398.25  5495.3 2397.77
  5516.8 2397.84  5904.9 2400.62  6003.0 2407.81  6065.4 2414.17  6095.5 2420.19
  6165.7 2452.71  6185.8 2464.86  6232.3 2470.95  6255.6 2471.15  6296.1 2475.49
#Mann=11,-1,0
  4591.7   0.035       0  4831.4    0.07       0  4873.7   0.035       0
  4982.3    0.16       0  5004.0    0.07       0  5040.0    0.16       0
  5229.0    0.07       0  5495.3    0.16       0  5516.8    0.07       0
  6003.0    0.16       0  6255.6    0.07       0
Bank Sta=5004,5040
Exp/Cntr=0.3,0.1

Type RM Length L Ch R = 1,303500,500,500,500
BEGIN DESCRIPTION:
Sweetwater Creek 605.0
END DESCRIPTION:
XS GIS Cut Line= 3
      1367705.01      6795788.00      1368692.23      6796025.97
      1369104.99      6796287.99
#Sta/Elev= 30
  3984.5 2444.46  4035.9 2436.41  4128.5 2426.46  4180.8 2413.11  4210.8 2409.78
  4282.8 2407.84  4301.4 2409.86  4395.9 2402.54  4529.7 2397.95  4797.9 2395.38
  4910.3 2395.31  4936.3 2388.05  4945.5 2386.79  4951.4 2382.57  4969.3 2377.82
  4970.2 2377.32  5005.4 2377.82  5011.2 2384.54  5032.3 2384.15  5068.8 2389.51
  5156.9 2389.99  5235.6 2385.93  5279.8 2387.94  5336.3 2387.11  5366.1 2386.03
  5381.3 2388.39  5444.9 2423.48  5453.4 2431.27  5460.1 2442.96  5488.9 2445.18
#Mann=7,-1,0
  3984.5    0.07       0  4797.9   0.035       0  4936.3    0.16       0
  4969.3    0.07       0  5005.4    0.16       0  5279.8    0.07       0
  5336.3    0.16       0
Bank Sta=4969.3,5005.4
Exp/Cntr=0.3,0.1

Type RM Length L Ch R = 1,303000,500,500,500
BEGIN DESCRIPTION:
Sweetwater Creek 604.0
END DESCRIPTION:
XS GIS Cut Line= 3
      1367655.02      6795788.01      1368655.86      6796507.12
      1368754.97      6796587.97
#Sta/Elev= 30
  3767.6 2451.36  3846.2 2441.04  3860.9 2436.91  3925.9 2430.10  3997.2 2415.58
  4018.0 2414.06  4032.8 2410.33  4144.5 2403.64  4314.1 2398.41  4397.4 2394.74
  4590.8 2392.99  4764.5 2393.10  4789.8 2391.42  4856.6 2384.67  4923.1 2382.37
  4963.4 2378.36  4992.9 2379.81  4995.6 2373.08  4996.4 2372.58  5032.0 2373.08
  5036.0 2386.90  5050.4 2396.73  5056.9 2405.99  5063.4 2410.58  5071.2 2411.63
  5077.7 2426.01  5085.6 2429.90  5092.0 2442.57  5106.4 2446.02  5127.9 2445.97
#Mann=8,-1,0
  3767.6    0.07       0  4144.5    0.16       0  4314.1    0.07       0
  4590.8   0.035       0  4789.8    0.16       0  4923.1    0.07       0
  4995.6    0.07       0  5032.0    0.07       0
Bank Sta=4995.6,5032
Exp/Cntr=0.3,0.1

Type RM Length L Ch R = 1,302500,500,500,500
BEGIN DESCRIPTION:
Sweetwater Creek 603.0
END DESCRIPTION:
XS GIS Cut Line= 3
      1367704.97      6796137.97      1368209.81      6796640.76
      1368605.03      6796888.02
#Sta/Elev= 30
  4287.5 2423.81  4330.0 2421.22  4429.0 2401.81  4471.4 2396.66  4575.7 2393.33
  4742.9 2390.40  4867.4 2388.12  4895.6 2385.83  4923.9 2377.76  4944.9 2376.75
  4987.6 2375.16  4989.9 2373.03  4990.8 2372.53  5026.3 2373.03  5096.5 2378.15
  5102.4 2376.02  5135.1 2376.44  5154.3 2375.99  5183.1 2382.54  5216.8 2394.45
  5248.6 2406.05  5254.5 2404.76  5264.0 2408.21  5269.9 2406.73  5285.2 2414.03
  5291.1 2412.46  5306.4 2415.88  5343.0 2432.79  5371.8 2439.51  5466.2 2449.13
#Mann=8,-1,0
  4287.5    0.16       0  4575.7   0.035       0  4742.9    0.16       0
  4944.9   0.035       0  4989.9   0.035       0  5026.3   0.035       0
  5135.1    0.16       0  5216.8    0.07       0
Bank Sta=4989.9,5026.3
Exp/Cntr=0.3,0.1

Type RM Length L Ch R = 1,302000,500,500,500
BEGIN DESCRIPTION:
Sweetwater Creek 602.0
END DESCRIPTION:
XS GIS Cut Line= 3
      1367405.00      6796388.00      1367905.01      6796900.49
      1368305.01      6797138.00
#Sta/Elev= 30
  4284.0 2431.20  4297.1 2427.53  4319.4 2420.15  4361.8 2415.46  4368.8 2417.43
  4489.1 2396.44  4545.7 2390.54  4701.3 2386.24  4920.5 2384.70  4934.6 2383.05
  4941.6 2379.15  4948.7 2378.59  4955.7 2369.26  4958.7 2368.06  4959.6 2367.56
  4995.3 2368.06  4996.4 2373.63  5011.6 2373.44  5034.9 2378.96  5063.8 2377.10
  5100.8 2380.26  5189.0 2380.27  5202.1 2380.30  5232.6 2385.33  5356.4 2391.90
  5407.0 2398.34  5436.0 2403.39  5451.6 2410.08  5457.4 2408.11  5465.2 2410.39
#Mann=6,-1,0
  4284.0   0.063       0  4297.1    0.16       0  4958.7    0.07       0
  4995.3    0.16       0  5189.0   0.035       0  5356.4    0.07       0
Bank Sta=4958.7,4995.3
Exp/Cntr=0.3,0.1

Type RM Length L Ch R = 1,301500,500,500,500
BEGIN DESCRIPTION:
Sweetwater Creek 601.0
END DESCRIPTION:
XS GIS Cut Line= 3
      1367155.02      6797038.01      1367647.26      6797247.35
      1368305.00      6797288.00
#Sta/Elev= 30
  4465.1 2414.27  4467.8 2414.27  4474.2 2406.50  4479.6 2403.61  4486.8 2396.93
  4508.7 2391.84  4671.5 2386.49  4716.4 2381.33  4812.5 2377.77  4861.4 2376.89
  4885.1 2379.58  4932.3 2375.56  4961.4 2375.70  4996.1 2367.47  5014.7 2367.41
  5049.6 2366.43  5050.5 2365.93  5086.2 2366.43  5087.2 2368.82  5097.9 2374.60
  5148.0 2374.72  5178.1 2382.34  5198.1 2384.33  5341.1 2384.94  5534.3 2392.12
  5549.4 2392.12  5580.9 2400.81  5608.9 2415.78  5628.9 2434.34  5659.0 2438.12
#Mann=9,-1,0
  4465.1    0.16       0  4716.4    0.07       0  4812.5    0.16       0
  5014.7    0.07       0  5049.6    0.07       0  5086.2    0.07       0
  5341.1   0.035       0  5534.3    0.16       0  5549.4    0.07       0
Bank Sta=5049.6,5086.2
Exp/Cntr=0.3,0.1

Type RM Length L Ch R = 1,301000,500,500,500
BEGIN DESCRIPTION:
Sweetwater Creek 600.0
END DESCRIPTION:
XS GIS Cut Line= 3
      1367055.02      6797588.00      1367406.89      6797636.54
      1368355.00      6797688.00
#Sta/Elev= 30
  4644.8 2431.27  4654.9 2433.24  4672.9 2429.80  4685.8 2427.75  4695.2 2421.44
  4705.3 2404.51  4715.4 2394.67  4752.7 2371.84  4776.0 2367.46  4856.8 2371.16
  4877.0 2368.22  4917.3 2369.82  4957.7 2367.66  4967.8 2365.47  4969.6 2362.24
  4970.5 2361.74  5006.3 2362.24  5008.1 2367.30  5038.2 2374.64  5121.3 2378.24
  5188.4 2381.99  5238.5 2379.99  5590.5 2381.09  5673.4 2383.95  5709.1 2388.11
  5764.8 2399.30  5819.3 2417.28  5839.3 2429.54  5855.8 2434.10  5949.5 2445.77
#Mann=7,-1,0
  4644.8    0.07       0  4672.9    0.16       0  4969.6    0.07       0
  5006.3    0.16       0  5121.3    0.07       0  5590.5   0.035       0
  5764.8    0.07       0
Bank Sta=4969.6,5006.3
Exp/Cntr=0.3,0.1

Type RM Length L Ch R = 1,300500,500,500,500
BEGIN DESCRIPTION:
Sweetwater Creek 599.0
END DESCRIPTION:
XS GIS Cut Line= 3
      1366955.05      6797938.01      1367149.62      6797986.82
      1368105.05      6797737.99
#Sta/Elev= 30
  4799.4 2442.74  4817.4 2436.60  4822.5 2437.69  4840.6 2432.78  4850.9 2420.51
  4858.5 2414.56  4871.5 2415.75  4881.8 2414.77  4892.1 2409.31  4899.7 2403.36
  4904.9 2402.36  4920.0 2390.99  4933.4 2381.31  4940.9 2374.15  4946.0 2374.43
  4954.0 2366.95  4963.7 2360.17  4964.6 2359.67  5000.4 2360.17  5012.9 2367.76
  5053.4 2371.07  5169.8 2374.50  5210.3 2373.59  5252.8 2374.82  5346.6 2377.76
  5463.9 2377.75  5634.5 2378.78  5877.4 2380.40  5956.3 2383.30  5987.3 2388.18
#Mann=8,-1,0
  4799.4    0.07       0  4920.0    0.16       0  4963.7    0.07       0
  5000.4    0.16       0  5252.8    0.07       0  5463.9    0.16       0
  5634.5    0.07       0  5877.4   0.035       0
Bank Sta=4963.7,5000.4
Exp/Cntr=0.3,0.1

Type RM Length L Ch R = 1,300000,500,500,500
BEGIN DESCRIPTION:
Sweetwater Creek 598.0
END DESCRIPTION:
XS GIS Cut Line= 3
      1367154.98      6798538.02      1367229.06      6798462.20
      1368154.97      6797888.02
#Sta/Elev= 30
  4894.0 2403.14  4901.1 2401.87  4908.1 2395.51  4913.4 2393.73  4922.2 2388.67
  4929.4 2390.24  4936.4 2388.48  4943.5 2391.09  4957.7 2388.83  4964.7 2383.04
  4967.6 2358.85  4968.5 2358.35  5004.3 2358.85  5021.1 2359.56  5057.7 2366.46
  5136.8 2365.61  5152.2 2367.09  5195.3 2364.25  5225.4 2372.76  5246.7 2373.46
  5611.0 2376.04  5631.6 2376.04  5724.5 2376.56  5973.7 2379.90  6024.0 2383.43
  6054.2 2390.63  6066.5 2390.28  6081.8 2393.50  6086.6 2399.06  6089.5 2399.06
#Mann=8,-1,0
  4894.0    0.07       0  4913.4    0.16       0  4967.6    0.07       0
  5004.3    0.16       0  5611.0    0.07       0  5631.6    0.16       0
  5724.5    0.07       0  5973.7   0.035       0
Bank Sta=4967.6,5004.3
Exp/Cntr=0.3,0.1

Type RM Length L Ch R = 1,299500,500,500,500
BEGIN DESCRIPTION:
Sweetwater Creek 597.0
END DESCRIPTION:
XS GIS Cut Line= 3
      1367205.02      6798887.99      1367576.83      6798787.67
      1368505.03      6798387.99
#Sta/Elev= 30
  4614.9 2405.07  4625.2 2406.06  4637.4 2401.22  4672.1 2372.78  4687.4 2366.69
  4739.2 2359.97  4786.7 2358.54  4822.3 2364.07  4826.6 2368.17  4830.6 2366.14
  4842.7 2364.17  4873.8 2368.11  4899.7 2367.23  4946.3 2358.25  5001.4 2357.01
  5002.3 2356.51  5038.1 2357.01  5042.1 2361.32  5090.2 2360.25  5106.9 2363.66
  5112.6 2367.88  5145.2 2370.52  5387.8 2370.09  5760.6 2378.81  5825.9 2395.21
  5873.0 2416.42  5896.5 2430.94  5912.4 2434.60  5972.5 2445.20  6010.6 2448.25
#Mann=9,-1,0
  4614.9    0.07       0  4822.3    0.16       0  4830.6    0.07       0
  5001.4    0.07       0  5038.1    0.07       0  5090.2    0.16       0
  5145.2    0.07       0  5760.6    0.16       0  5912.4    0.07       0
Bank Sta=5001.4,5038.1
Exp/Cntr=0.3,0.1

Type RM Length L Ch R = 1,299000,500,500,500
BEGIN DESCRIPTION:
Sweetwater Creek 596.0
END DESCRIPTION:
XS GIS Cut Line= 3
      1367404.97      6799388.02      1367897.38      6799130.02
      1368304.98      6798638.03
#Sta/Elev= 30
  4444.1 2412.46  4458.0 2410.87  4480.0 2403.06  4496.5 2394.71  4518.5 2387.02
  4546.2 2379.73  4557.0 2379.10  4590.9 2372.72  4639.0 2369.47  4681.2 2368.67
  4802.3 2371.98  4815.6 2371.65  4860.3 2372.06  4895.7 2368.08  4904.4 2368.65
  4908.5 2366.85  4932.1 2361.14  4970.6 2355.79  4970.9 2352.49  4971.9 2351.99
  5014.4 2352.49  5014.5 2353.77  5028.6 2354.26  5070.4 2364.14  5106.5 2367.33
  5320.7 2367.73  5418.2 2370.94  5547.1 2372.24  5596.6 2374.10  5638.9 2377.67
#Mann=8,-1,0
  4444.1    0.07       0  4639.0   0.035       0  4802.3    0.16       0
  4815.6    0.07       0  4908.5    0.16       0  4970.9    0.07       0
  5014.4    0.16       0  5320.7    0.07       0
Bank Sta=4970.9,5014.4
Exp/Cntr=0.3,0.1

Type RM Length L Ch R = 1,298500,500,500,500
BEGIN DESCRIPTION:
Sweetwater Creek 595.0
END DESCRIPTION:
XS GIS Cut Line= 3
      1368204.99      6799538.01      1368268.62      6799451.99
      1368654.99      6798938.02
#Sta/Elev= 30
  4893.0 2364.80  4896.1 2364.80  4921.2 2354.42  4950.4 2353.08  4971.3 2343.26
  4993.3 2342.59  4994.3 2342.09  5036.9 2342.59  5042.5 2357.43  5050.5 2358.72
  5265.0 2365.06  5379.6 2372.48  5385.8 2374.43  5435.8 2379.29  5500.4 2383.53
  5506.6 2385.70  5514.9 2384.82  5529.5 2388.03  5535.8 2391.53  5550.3 2391.53
  5571.2 2397.70  5579.5 2397.47  5585.7 2400.48  5600.3 2400.21  5606.6 2403.36
  5614.9 2402.81  5621.2 2406.20  5629.5 2406.15  5635.7 2410.31  5643.0 2409.34
#Mann=3,-1,0
  4893.0    0.07       0  4993.3    0.07       0  5036.9    0.16       0
Bank Sta=4993.3,5036.9
Exp/Cntr=0.3,0.1

Type RM Length L Ch R = 1,298000,500,500,500
BEGIN DESCRIPTION:
Sweetwater Creek 594.0
END DESCRIPTION:
XS GIS Cut Line= 3
      1368205.04      6799788.01      1368562.45      6799835.85
      1368955.00      6799488.00
#Sta/Elev= 30
  4639.4 2363.53  4720.1 2361.53  4841.1 2361.93  4851.2 2360.85  4871.4 2354.00
  4891.6 2350.79  4934.4 2350.11  4962.2 2342.07  4977.0 2340.65  4978.0 2340.15
  5020.6 2340.65  5058.8 2347.75  5099.2 2357.11  5191.2 2355.20  5227.9 2357.30
  5319.2 2359.27  5354.3 2368.29  5390.3 2383.08  5404.2 2385.76  5413.1 2390.87
  5439.6 2402.40  5446.3 2403.09  5453.8 2406.65  5461.3 2407.30  5468.0 2412.00
  5474.7 2412.39  5482.3 2416.47  5488.9 2417.04  5510.7 2426.56  5524.5 2429.69
#Mann=8,-1,0
  4639.4   0.035       0  4934.4    0.07       0  4977.0    0.07       0
  5020.6    0.07       0  5058.8   0.035       0  5227.9    0.16       0
  5413.1   0.035       0  5461.3    0.07       0
Bank Sta=4977,5020.6
Exp/Cntr=0.3,0.1

Type RM Length L Ch R = 1,297500,500,500,500
BEGIN DESCRIPTION:
Sweetwater Creek 593.0
END DESCRIPTION:
XS GIS Cut Line= 3
      1368104.99      6800138.00      1368805.22      6800223.25
      1369055.05      6800187.99
#Sta/Elev= 30
  4294.6 2363.38  4332.9 2363.82  4395.3 2362.27  4419.6 2360.96  4455.8 2354.98
  4475.9 2354.02  4546.5 2354.47  4617.0 2357.45  4737.9 2357.25  4751.3 2353.04
  4758.0 2348.43  4768.1 2346.02  4788.2 2346.13  4808.4 2351.13  4848.7 2345.31
  4878.9 2346.11  4899.0 2344.49  4939.3 2345.02  4959.5 2340.94  4987.1 2339.85
  4988.1 2339.35  5032.7 2339.85  5043.5 2342.63  5060.4 2346.86  5069.4 2351.24
  5074.4 2352.26  5145.6 2351.42  5171.5 2364.49  5214.4 2366.46  5252.3 2367.58
#Mann=5,-1,0
  4294.6    0.07       0  4987.1    0.07       0  5032.7    0.07       0
  5043.5   0.035       0  5214.4    0.16       0
Bank Sta=4987.1,5032.7
Exp/Cntr=0.3,0.1

Type RM Length L Ch R = 1,297000,500,500,500
BEGIN DESCRIPTION:
Sweetwater Creek 592.0
END DESCRIPTION:
XS GIS Cut Line= 3
      1368155.02      6800338.01      1368484.05      6800537.53
      1368604.97      6800637.98
#Sta/Elev= 30
  4615.2 2359.91  4625.6 2358.59  4644.3 2356.91  4650.3 2353.26  4659.8 2350.11
  4673.7 2347.48  4686.9 2346.87  4745.1 2346.85  4860.0 2350.20  4884.2 2350.46
  4913.8 2353.70  4929.2 2353.52  4950.6 2351.75  4966.0 2347.00  4971.9 2341.92
  4974.8 2335.85  4975.8 2335.35  5020.4 2335.85  5022.5 2336.59  5051.1 2337.77
  5079.2 2344.31  5086.3 2347.29  5092.8 2346.41  5114.9 2348.58  5121.4 2347.52
  5129.2 2348.34  5135.7 2350.61  5143.6 2355.18  5150.1 2356.79  5157.2 2357.17
#Mann=5,-1,0
  4615.2    0.07       0  4625.6    0.16       0  4860.0    0.07       0
  4974.8    0.07       0  5020.4    0.07       0
Bank Sta=4974.8,5020.4
Exp/Cntr=0.3,0.1

Type RM Length L Ch R = 1,296500,500,500,500
BEGIN DESCRIPTION:
Sweetwater Creek 591.0
END DESCRIPTION:
XS GIS Cut Line= 3
      1367855.00      6800838.00      1368200.15      6800889.00
      1369155.01      6800638.00
#Sta/Elev= 30
  4651.1 2367.87  4671.3 2367.78  4700.9 2363.61  4782.5 2359.53  4833.1 2354.36
  4889.6 2346.22  4924.0 2336.73  4951.8 2334.62  4952.8 2334.12  4997.4 2334.62
  4999.9 2338.27  5022.1 2339.15  5056.7 2338.61  5077.4 2336.61  5102.8 2337.40
  5118.7 2340.74  5129.1 2341.10  5218.6 2340.49  5273.8 2342.56  5299.3 2344.59
  5334.5 2353.03  5346.2 2352.27  5374.8 2355.53  5439.3 2356.26  5480.6 2358.82
  5725.3 2360.76  5873.6 2369.87  5902.7 2373.66  5942.1 2376.54  5987.3 2383.20
#Mann=7,-1,0
  4651.1    0.16       0  4700.9    0.07       0  4951.8    0.07       0
  4997.4    0.07       0  5725.3   0.035       0  5902.7    0.16       0
  5942.1    0.07       0
Bank Sta=4951.8,4997.4
Exp/Cntr=0.3,0.1

Type RM Length L Ch R = 1,296000,500,500,500
BEGIN DESCRIPTION:
Sweetwater Creek 590.0
END DESCRIPTION:
XS GIS Cut Line= 3
      1368255.00      6801538.03      1368296.10      6801280.49
      1368554.98      6800938.03
#Sta/Elev= 30
  4739.2 2362.88  4759.5 2363.45  4772.8 2361.61  4820.2 2346.16  4840.5 2341.77
  4860.8 2339.38  4881.0 2334.20  4959.1 2333.73  4959.4 2332.65  4960.4 2332.15
  5005.2 2332.65  5028.8 2336.83  5051.6 2337.79  5072.4 2337.01  5078.7 2338.40
  5087.0 2336.70  5128.6 2336.93  5157.8 2338.48  5166.1 2337.75  5178.6 2339.76
  5207.7 2337.11  5222.3 2340.10  5265.9 2338.99  5286.8 2342.40  5293.0 2348.30
  5301.3 2350.00  5307.6 2353.00  5320.9 2353.31  5406.1 2354.09  5429.3 2354.29
#Mann=5,-1,0
  4739.2    0.07       0  4959.4    0.07       0  5005.2    0.07       0
  5320.9    0.16       0  5406.1    0.07       0
Bank Sta=4959.4,5005.2
Exp/Cntr=0.3,0.1

Type RM Length L Ch R = 1,295500,500,500,500
BEGIN DESCRIPTION:
Sweetwater Creek 589.0
END DESCRIPTION:
XS GIS Cut Line= 3
      1368455.02      6801687.99      1368631.24      6801588.03
      1368905.02      6801237.98
#Sta/Elev= 30
  4797.4 2354.57  4864.5 2353.87  4870.2 2352.26  4886.1 2351.76  4891.8 2346.83
  4900.9 2345.02  4913.5 2337.50  4929.4 2336.27  4951.0 2332.54  4988.5 2331.60
  4993.7 2330.51  4994.7 2330.01  5039.5 2330.51  5045.6 2332.34  5060.0 2333.49
  5102.5 2333.67  5116.1 2336.37  5130.6 2335.67  5145.1 2338.20  5152.4 2342.26
  5165.9 2345.31  5202.9 2345.72  5223.7 2343.81  5273.5 2344.25  5366.6 2340.74
  5387.4 2344.11  5403.1 2348.94  5416.3 2352.97  5430.8 2355.13  5444.4 2355.20
#Mann=5,-1,0
  4797.4    0.07       0  4993.7    0.07       0  5039.5    0.07       0
  5102.5    0.16       0  5403.1    0.07       0
Bank Sta=4993.7,5039.5
Exp/Cntr=0.3,0.1

Type RM Length L Ch R = 1,295000,500,500,500
BEGIN DESCRIPTION:
Sweetwater Creek 588.0
END DESCRIPTION:
XS GIS Cut Line= 3
      1368454.97      6801838.00      1368963.32      6801894.67
      1369354.96      6801987.99
#Sta/Elev= 30
  4488.5 2353.45  4805.0 2348.01  4840.7 2337.49  4860.8 2337.15  4890.3 2332.02
  4991.6 2331.75  5030.2 2329.31  5031.2 2328.81  5076.0 2329.31  5079.0 2331.43
  5145.6 2329.64  5163.2 2332.36  5168.4 2331.26  5177.0 2334.28  5205.3 2342.89
  5210.5 2338.76  5217.6 2340.44  5238.2 2346.55  5247.5 2352.16  5252.6 2348.86
  5258.7 2356.24  5269.0 2361.41  5279.3 2364.84  5320.4 2370.92  5336.9 2379.30
  5371.8 2389.96  5379.1 2397.04  5384.1 2394.45  5400.1 2405.59  5402.6 2405.59
#Mann=5,-1,0
  4488.5    0.07       0  5030.2    0.07       0  5076.0    0.07       0
  5177.0   0.035       0  5379.1    0.16       0
Bank Sta=5030.2,5076
Exp/Cntr=0.3,0.1

Type RM Length L Ch R = 1,294500,500,500,500
BEGIN DESCRIPTION:
Sweetwater Creek 587.0
END DESCRIPTION:
XS GIS Cut Line= 3
      1368555.02      6802088.01      1369054.73      6802306.02
      1369454.99      6802238.00
#Sta/Elev= 30
  4454.8 2349.67  4597.2 2349.02  4651.2 2339.88  4714.3 2339.92  4743.1 2345.81
  4782.1 2344.82  4842.2 2339.34  4894.5 2330.81  4956.7 2330.11  4964.8 2329.50
  4965.2 2326.96  4966.2 2326.46  5011.1 2326.96  5016.8 2329.56  5071.4 2329.75
  5152.4 2329.73  5172.7 2337.49  5192.5 2350.40  5197.6 2348.77  5203.1 2356.00
  5213.3 2364.34  5223.4 2368.07  5243.7 2369.43  5273.2 2386.17  5313.1 2414.14
  5318.1 2413.10  5324.9 2420.07  5345.2 2433.22  5373.3 2445.41  5406.0 2449.43
#Mann=5,-1,0
  4454.8    0.07       0  4965.2    0.07       0  5011.1    0.07       0
  5071.4   0.035       0  5273.2    0.16       0
Bank Sta=4965.2,5011.1
Exp/Cntr=0.3,0.1

Type RM Length L Ch R = 1,294000,500,500,500
BEGIN DESCRIPTION:
Sweetwater Creek 586.0
END DESCRIPTION:
XS GIS Cut Line= 3
      1368105.01      6802088.00      1369105.09      6802789.88
      1369505.02      6802587.99
#Sta/Elev= 30
  3778.2 2371.56  3806.5 2373.35  4024.5 2352.83  4544.0 2343.68  4624.9 2345.20
  4743.7 2341.44  4854.1 2339.99  4949.1 2328.32  4953.1 2324.97  4954.1 2324.47
  4999.0 2324.97  5000.0 2327.46  5006.6 2327.26  5038.3 2325.32  5055.0 2332.43
  5077.3 2335.12  5119.1 2335.15  5156.7 2337.66  5179.1 2345.09  5256.4 2358.17
  5291.2 2359.82  5344.1 2371.62  5350.4 2370.69  5372.7 2376.21  5395.0 2389.14
  5411.7 2402.14  5417.3 2401.52  5434.0 2412.83  5439.6 2412.34  5448.0 2417.24
#Mann=10,-1,0
  3778.2    0.16       0  4024.5    0.07       0  4544.0    0.16       0
  4743.7    0.07       0  4953.1    0.07       0  4999.0    0.07       0
  5006.6    0.16       0  5119.1   0.035       0  5256.4    0.07       0
  5344.1    0.16       0
Bank Sta=4953.1,4999
Exp/Cntr=0.3,0.1

Type RM Length L Ch R = 1,293500,500,500,500
BEGIN DESCRIPTION:
Sweetwater Creek 585.0
END DESCRIPTION:
XS GIS Cut Line= 3
      1368504.99      6802737.99      1369005.11      6803257.62
      1369255.00      6803188.00
#Sta/Elev= 30
  4278.8 2349.10  4335.3 2348.98  4524.7 2345.37  4540.6 2345.67  4561.7 2343.99
  4611.3 2343.19  4653.5 2340.34  4660.7 2340.98  4681.8 2339.56  4771.1 2337.96
  4887.1 2336.89  4894.1 2334.59  4901.3 2334.17  4922.4 2330.13  4929.6 2330.34
  4943.7 2327.41  4986.2 2327.22  4987.3 2322.87  4988.3 2322.37  5033.2 2322.87
  5041.4 2326.56  5062.2 2326.15  5082.9 2329.69  5089.9 2332.04  5095.1 2331.27
  5124.1 2339.50  5129.3 2339.21  5163.5 2342.89  5200.2 2345.39  5259.4 2351.17
#Mann=7,-1,0
  4278.8    0.16       0  4524.7    0.07       0  4771.1    0.16       0
  4887.1    0.07       0  4987.3    0.07       0  5033.2    0.07       0
  5200.2   0.035       0
Bank Sta=4987.3,5033.2
Exp/Cntr=0.3,0.1

Type RM Length L Ch R = 1,293000,500,500,500
BEGIN DESCRIPTION:
Sweetwater Creek 584.0
END DESCRIPTION:
XS GIS Cut Line= 3
      1368455.04      6803638.01      1368809.35      6803683.38
      1369204.96      6803638.00
#Sta/Elev= 30
  4642.8 2347.59  4652.8 2346.22  4753.7 2341.79  4764.8 2341.80  4878.9 2335.72
  4914.1 2334.04  4919.1 2332.46  4935.1 2331.01  4945.2 2327.89  4965.4 2323.75
  4993.8 2324.09  5002.0 2322.40  5002.5 2320.85  5003.5 2320.35  5048.2 2320.35
  5049.2 2320.85  5056.0 2322.69  5066.1 2323.53  5076.1 2326.46  5086.1 2327.65
  5091.2 2326.99  5096.3 2328.69  5126.5 2328.80  5136.5 2329.59  5156.7 2333.43
  5175.3 2335.63  5196.9 2334.40  5237.2 2337.87  5327.1 2341.22  5398.2 2343.91
#Mann=5,-1,0
  4642.8    0.16       0  4878.9    0.07       0  5002.5    0.07       0
  5049.2    0.07       0  5327.1   0.035       0
Bank Sta=5002.5,5049.2
Exp/Cntr=0.3,0.1

Type RM Length L Ch R = 1,292500,500,500,500
BEGIN DESCRIPTION:
Sweetwater Creek 583.0
END DESCRIPTION:
XS GIS Cut Line= 3
      1368654.98      6804238.02      1368713.86      6804145.58
      1369105.03      6803787.97
#Sta/Elev= 30
  4890.4 2340.07  4934.4 2338.31  4940.4 2337.09  4949.7 2337.82  4955.6 2334.42
  4970.8 2332.38  4973.0 2318.89  4974.0 2318.39  5019.9 2318.89  5020.3 2320.15
  5027.7 2321.42  5048.6 2323.49  5077.0 2321.41  5105.4 2321.94  5140.5 2321.15
  5147.9 2320.06  5162.1 2322.13  5168.9 2321.66  5176.3 2324.75  5183.1 2322.89
  5190.5 2325.26  5197.2 2323.30  5246.6 2323.83  5260.8 2325.21  5268.2 2330.43
  5274.9 2331.61  5317.5 2331.75  5374.2 2335.25  5462.6 2337.42  5530.0 2340.06
#Mann=4,-1,0
  4890.4    0.07       0  4973.0    0.07       0  5019.9    0.07       0
  5462.6   0.035       0
Bank Sta=4973,5019.9
Exp/Cntr=0.3,0.1
