HEC-RAS study Sweetwater Creek.prj: Sweetwater Creek Base Level Engineering

--- Sweetwater Creek.g01 (geometry) --- (continued)

Type RM Length L Ch R = 1,266500,500,500,500
BEGIN DESCRIPTION:
Sweetwater Creek 531.0
END DESCRIPTION:
XS GIS Cut Line= 3
      1371805.03      6824138.00      1372139.47      6824172.37
      1372555.02      6824438.01
#Sta/Elev= 30
  4663.8 2235.36  4834.7 2234.33  4854.8 2232.44  4909.2 2231.62  4928.1 2228.04
  4982.1 2213.64  4982.7 2212.64  5006.2 2213.64  5022.0 2213.76  5037.3 2217.44
  5043.2 2215.86  5052.5 2217.52  5058.4 2216.92  5088.9 2222.92  5094.8 2221.84
  5110.0 2227.10  5146.4 2227.94  5167.5 2215.22  5173.5 2214.42  5182.7 2215.01
  5215.7 2223.95  5267.7 2228.17  5297.8 2223.34  5318.9 2232.03  5355.3 2231.51
  5362.6 2235.63  5391.7 2244.30  5398.2 2248.30  5449.2 2254.18  5493.2 2263.56
#Mann=5,-1,0
  4663.8    0.07       0  4928.1    0.16       0  4982.1    0.07       0
  5006.2    0.16       0  5215.7    0.07       0
Bank Sta=4982.1,5006.2
Exp/Cntr=0.3,0.1

Type RM Length L Ch R = 1,266000,500,500,500
BEGIN DESCRIPTION:
Sweetwater Creek 530.0
END DESCRIPTION:
XS GIS Cut Line= 3
      1371805.02      6824338.02      1372004.34      6824543.40
      1372104.98      6824637.98
#Sta/Elev= 30
  4713.8 2233.70  4733.0 2234.03  4742.0 2234.14  4749.1 2233.07  4777.4 2233.01
  4848.2 2230.50  4911.7 2226.37  4918.9 2226.57  4947.2 2223.09  4961.3 2220.07
  4968.3 2220.24  4975.5 2218.34  4982.5 2218.56  4989.6 2215.18  4990.8 2212.50
  4991.3 2211.50  5008.6 2211.50  5009.0 2212.50  5010.9 2213.53  5025.1 2214.67
  5031.9 2215.91  5060.2 2217.43  5067.5 2219.40  5074.4 2235.00  5081.7 2247.59
  5088.6 2251.52  5095.9 2253.60  5102.7 2253.51  5110.0 2254.35  5138.1 2255.79
#Mann=4,-1,0
  4713.8   0.035       0  4733.0    0.07       0  4990.8    0.07       0
  5009.0    0.07       0
Bank Sta=4990.8,5009
Exp/Cntr=0.3,0.1

Type RM Length L Ch R = 1,265500,500,500,500
BEGIN DESCRIPTION:
Sweetwater Creek 529.0
END DESCRIPTION:
XS GIS Cut Line= 3
      1370855.05      6824937.99      1371699.87      6824739.18
      1372105.00      6825138.00
#Sta/Elev= 30
  4132.1 2273.20  4190.5 2257.58  4245.7 2252.04  4275.9 2239.09  4288.1 2237.56
  4409.4 2231.63  4573.8 2231.67  4638.4 2227.60  4686.8 2224.07  4722.1 2212.58
  4799.8 2230.29  4843.1 2230.08  4882.0 2230.22  4933.8 2221.80  4939.1 2217.62
  4944.2 2219.49  4964.2 2211.47  4977.6 2210.69  4978.2 2209.69  5001.9 2210.69
  5002.8 2216.21  5088.5 2220.46  5198.3 2224.02  5232.1 2228.32  5306.8 2238.95
  5328.1 2249.73  5420.0 2264.33  5455.4 2274.77  5552.6 2292.98  5568.5 2294.20
#Mann=11,-1,0
  4132.1   0.035       0  4190.5    0.07       0  4638.4    0.16       0
  4843.1    0.07       0  4933.8    0.16       0  4977.6    0.07       0
  5001.9    0.16       0  5088.5    0.07       0  5198.3    0.16       0
  5232.1    0.07       0  5552.6   0.035       0
Bank Sta=4977.6,5001.9
Exp/Cntr=0.3,0.1

Type RM Length L Ch R = 1,265000,500,500,500
BEGIN DESCRIPTION:
Sweetwater Creek 528.0
END DESCRIPTION:
XS GIS Cut Line= 3
      1371054.97      6825438.01      1371554.91      6825187.04
      1371955.02      6825138.00
#Sta/Elev= 30
  4440.6 2243.18  4443.4 2243.18  4449.0 2239.93  4454.6 2239.58  4463.0 2235.90
  4471.3 2234.18  4493.7 2231.68  4538.3 2229.08  4583.0 2228.25  4722.6 2228.49
  4744.9 2229.55  4878.9 2229.04  4923.6 2225.10  4938.4 2218.89  4955.3 2215.85
  4977.7 2213.78  4987.9 2211.35  4988.4 2210.35  5006.0 2210.35  5006.5 2211.35
  5010.2 2214.64  5050.5 2217.20  5080.7 2222.89  5115.7 2223.05  5191.5 2228.39
  5221.7 2228.36  5301.6 2233.67  5342.6 2237.75  5372.9 2249.55  5403.1 2256.47
#Mann=5,-1,0
  4440.6    0.07       0  4938.4    0.16       0  4987.9    0.07       0
  5006.5    0.16       0  5301.6    0.07       0
Bank Sta=4987.9,5006.5
Exp/Cntr=0.3,0.1

Type RM Length L Ch R = 1,264500,500,500,500
BEGIN DESCRIPTION:
Sweetwater Creek 527.0
END DESCRIPTION:
XS GIS Cut Line= 3
      1370904.99      6825438.00      1371774.36      6825557.12
      1372005.03      6825487.99
#Sta/Elev= 30
  4122.5 2269.25  4179.5 2269.81  4203.3 2270.47  4213.4 2268.67  4253.7 2252.17
  4263.8 2249.53  4284.0 2239.83  4302.9 2234.18  4308.0 2234.71  4324.4 2231.18
  4405.1 2227.41  4626.4 2228.58  4687.7 2228.63  4697.8 2226.18  4751.0 2225.51
  4967.5 2212.07  4990.5 2212.91  4997.2 2208.56  4997.6 2207.56  5015.7 2208.56
  5021.5 2208.56  5042.4 2220.72  5048.4 2225.73  5094.6 2230.57  5119.8 2231.45
  5145.5 2234.90  5158.1 2239.19  5178.1 2253.56  5185.9 2256.44  5240.8 2256.85
#Mann=6,-1,0
  4122.5   0.035       0  4179.5    0.07       0  4626.4    0.16       0
  4997.2    0.07       0  5015.7    0.16       0  5145.5    0.07       0
Bank Sta=4997.2,5015.7
Exp/Cntr=0.3,0.1

Type RM Length L Ch R = 1,264000,500,500,500
BEGIN DESCRIPTION:
Sweetwater Creek 526.0
END DESCRIPTION:
XS GIS Cut Line= 3
      1371205.02      6826537.98      1371886.75      6826019.98
      1372305.03      6825988.00
#Sta/Elev= 30
  4143.8 2259.31  4146.9 2259.31  4157.3 2248.98  4165.6 2246.67  4221.8 2245.24
  4250.9 2229.01  4303.2 2223.25  4376.6 2221.88  4439.3 2224.70  4518.0 2225.44
  4645.1 2225.27  4751.6 2226.23  4772.2 2226.10  4849.8 2225.90  4864.4 2224.42
  4878.9 2219.20  4914.3 2215.45  4928.8 2211.13  4978.7 2211.39  4988.7 2205.40
  4989.2 2204.40  5007.3 2205.40  5008.3 2208.09  5048.4 2222.72  5249.0 2233.24
  5269.0 2236.18  5299.1 2245.04  5319.2 2247.17  5389.4 2255.11  5419.5 2260.90
#Mann=11,-1,0
  4143.8    0.07       0  4303.2    0.16       0  4376.6    0.07       0
  4439.3    0.16       0  4518.0    0.07       0  4645.1    0.16       0
  4751.6    0.07       0  4772.2    0.16       0  4988.7    0.07       0
  5007.3    0.16       0  5319.2    0.07       0
Bank Sta=4988.7,5007.3
Exp/Cntr=0.3,0.1

Type RM Length L Ch R = 1,263500,500,500,500
BEGIN DESCRIPTION:
Sweetwater Creek 525.0
END DESCRIPTION:
XS GIS Cut Line= 3
      1371554.99      6826888.01      1372038.62      6826471.91
      1372454.98      6826138.02
#Sta/Elev= 30
  4362.0 2230.45  4365.3 2230.45  4369.2 2226.30  4383.4 2222.33  4489.8 2219.30
  4544.5 2219.90  4581.6 2220.74  4688.5 2221.67  4794.9 2224.25  4836.9 2223.16
  4865.1 2221.58  4915.6 2215.56  4936.4 2214.96  4950.7 2210.82  4971.6 2210.21
  4986.5 2205.62  4986.9 2204.62  5005.0 2205.62  5008.0 2210.88  5021.0 2212.08
  5043.2 2217.21  5156.8 2223.12  5200.3 2223.84  5328.1 2228.11  5355.3 2232.36
  5384.1 2242.85  5483.3 2254.20  5512.1 2259.80  5520.1 2263.45  5533.7 2266.72
#Mann=7,-1,0
  4362.0    0.07       0  4544.5    0.16       0  4581.6    0.07       0
  4688.5    0.16       0  4986.5    0.07       0  5005.0    0.16       0
  5200.3    0.07       0
Bank Sta=4986.5,5005
Exp/Cntr=0.3,0.1

Type RM Length L Ch R = 1,263000,500,500,500
BEGIN DESCRIPTION:
Sweetwater Creek 524.0
END DESCRIPTION:
XS GIS Cut Line= 3
      1371805.01      6827187.99      1372158.31      6826934.91
      1372554.98      6826438.02
#Sta/Elev= 30
  4565.4 2248.62  4568.5 2248.62  4593.6 2230.96  4608.4 2223.04  4629.3 2218.02
  4677.7 2217.16  4795.1 2218.48  4816.0 2220.56  4937.6 2215.92  4981.8 2210.91
  4994.9 2206.69  4995.8 2200.34  4996.3 2199.34  5014.4 2200.34  5031.4 2203.61
  5037.8 2206.91  5081.0 2207.05  5109.9 2210.95  5116.3 2214.50  5137.1 2219.00
  5180.3 2217.61  5215.5 2220.61  5237.9 2219.33  5354.1 2221.30  5436.5 2222.01
  5550.2 2226.91  5564.6 2229.96  5593.4 2242.10  5614.2 2246.43  5635.8 2248.04
#Mann=5,-1,0
  4565.4    0.07       0  4677.7    0.16       0  4995.8    0.07       0
  5014.4    0.16       0  5354.1    0.07       0
Bank Sta=4995.8,5014.4
Exp/Cntr=0.3,0.1

Type RM Length L Ch R = 1,262500,500,500,500
BEGIN DESCRIPTION:
Sweetwater Creek 523.0
END DESCRIPTION:
XS GIS Cut Line= 3
      1371905.01      6827488.00      1372256.39      6827375.65
      1373128.27      6826954.19
#Sta/Elev= 30
  4631.1 2237.19  4633.7 2237.19  4647.2 2229.73  4652.4 2229.89  4679.3 2221.13
  4711.5 2216.58  4795.2 2216.39  4893.6 2218.36  4956.5 2214.85  4967.0 2211.16
  4974.1 2206.64  4979.3 2200.99  4987.1 2198.33  4987.6 2197.33  5005.7 2198.33
  5010.6 2204.69  5121.6 2215.26  5168.8 2219.13  5214.9 2219.43  5365.0 2219.99
  5564.9 2226.89  5722.2 2230.20  5739.2 2230.28  5753.2 2227.90  5784.4 2235.52
  5829.6 2239.12  5857.8 2244.81  5874.8 2250.23  5942.6 2256.22  5968.4 2255.91
#Mann=7,-1,0
  4631.1    0.07       0  4795.2    0.16       0  4987.1    0.07       0
  5005.7    0.16       0  5121.6    0.07       0  5214.9    0.16       0
  5753.2    0.07       0
Bank Sta=4987.1,5005.7
Exp/Cntr=0.3,0.1

Type RM Length L Ch R = 1,262000,500,500,500
BEGIN DESCRIPTION:
Sweetwater Creek 522.0
END DESCRIPTION:
XS GIS Cut Line= 3
      1371905.03      6827588.01      1372554.11      6827750.88
      1373181.25      6827507.80
#Sta/Elev= 30
  4330.8 2246.29  4402.9 2218.73  4467.9 2214.47  4591.8 2216.17  4761.2 2217.14
  4856.6 2212.60  4883.9 2207.15  4889.1 2208.47  4971.4 2202.62  4990.1 2196.76
  4990.5 2195.76  5008.6 2196.76  5019.4 2207.05  5024.8 2206.33  5033.1 2212.64
  5073.9 2216.46  5327.1 2219.26  5441.4 2222.90  5483.6 2228.02  5490.6 2231.05
  5495.9 2230.14  5515.1 2238.61  5520.5 2237.08  5526.5 2242.33  5543.6 2250.53
  5550.4 2249.57  5569.4 2255.14  5604.9 2256.35  5612.3 2258.84  5672.6 2260.28
#Mann=7,-1,0
  4330.8    0.07       0  4467.9    0.16       0  4591.8    0.12       0
  4761.2    0.16       0  4990.1    0.07       0  5008.6    0.16       0
  5543.6    0.07       0
Bank Sta=4990.1,5008.6
Exp/Cntr=0.3,0.1

Type RM Length L Ch R = 1,261500,500,500,500
BEGIN DESCRIPTION:
Sweetwater Creek 521.0
END DESCRIPTION:
XS GIS Cut Line= 3
      1371854.99      6827637.99      1372705.18      6828181.57
      1372954.99      6828437.99
#Sta/Elev= 30
  3990.9 2248.36  4019.7 2245.99  4050.1 2236.16  4062.1 2228.65  4098.3 2217.44
  4185.6 2213.46  4397.1 2217.01  4650.0 2216.14  4799.5 2211.22  4873.9 2209.90
  4889.2 2205.09  4952.6 2201.93  4985.6 2195.88  4986.1 2194.88  5004.2 2195.88
  5004.5 2201.85  5039.7 2212.11  5046.9 2211.05  5068.0 2216.34  5110.5 2217.04
  5117.6 2215.28  5202.5 2220.51  5209.5 2224.89  5216.6 2225.73  5248.2 2238.19
  5259.1 2243.90  5266.1 2250.47  5280.2 2255.19  5308.5 2258.06  5358.0 2258.22
#Mann=8,-1,0
  3990.9    0.07       0  4185.6    0.16       0  4397.1    0.12       0
  4650.0    0.16       0  4799.5    0.12       0  4985.6    0.07       0
  5004.2    0.12       0  5248.2    0.07       0
Bank Sta=4985.6,5004.2
Exp/Cntr=0.3,0.1

Type RM Length L Ch R = 1,261000,500,500,500
BEGIN DESCRIPTION:
Sweetwater Creek 520.0
END DESCRIPTION:
XS GIS Cut Line= 4
      1370164.54      6828573.98      1372257.53      6828530.23
      1372484.89      6828587.46      1372905.03      6828688.01
#Sta/Elev= 30
  2672.1 2241.24  2977.7 2231.05  3049.2 2230.54  3132.7 2226.15  3232.7 2226.73
  3272.7 2242.86  3292.7 2239.35  3312.7 2227.19  3332.7 2225.38  3362.7 2243.75
  3382.7 2244.61  3512.7 2238.48  3702.8 2215.57  3832.8 2219.16  4022.9 2213.86
  4386.4 2212.11  4880.4 2213.69  4936.9 2213.52  4978.0 2198.81  4983.2 2192.89
  4995.5 2191.39  4996.1 2190.39  5020.3 2191.39  5024.8 2197.58  5264.7 2220.89
  5282.2 2223.02  5318.9 2235.48  5339.4 2250.49  5360.0 2257.40  5432.0 2258.15
#Mann=8,-1,0
  2672.1    0.07       0  2977.7   0.035       0  3049.2    0.07       0
  4386.4    0.16       0  4880.4    0.12       0  4995.5    0.07       0
  5020.3    0.12       0  5264.7    0.07       0
Bank Sta=4995.5,5020.3
Exp/Cntr=0.3,0.1

Type RM Length L Ch R = 1,260500,500,500,500
BEGIN DESCRIPTION:
Sweetwater Creek 519.0
END DESCRIPTION:
XS GIS Cut Line= 3
      1370186.98      6828833.30      1372271.37      6828994.15
      1372777.12      6828977.82
#Sta/Elev= 30
  2926.3 2243.09  3205.1 2227.01  3516.1 2218.38  3576.8 2218.25  3596.3 2221.80
  3626.4 2216.48  3793.4 2211.93  3877.1 2210.49  3987.5 2214.21  4130.5 2214.47
  4595.6 2210.45  4884.2 2211.74  4960.4 2212.36  4980.4 2205.22  4990.4 2196.45
  4991.8 2189.51  4992.3 2188.51  5010.4 2189.51  5010.5 2196.08  5016.2 2198.52
  5110.6 2198.94  5129.9 2200.91  5160.6 2207.29  5260.6 2209.72  5359.7 2216.08
  5420.7 2223.06  5450.7 2232.79  5490.8 2253.55  5517.7 2256.64  5522.9 2256.72
#Mann=11,-1,0
  2926.3    0.07       0  3793.4   0.035       0  4130.5    0.07       0
  4595.6    0.16       0  4884.2    0.12       0  4991.8    0.07       0
  5010.4    0.12       0  5129.9    0.16       0  5260.6    0.12       0
  5359.7    0.07       0  5517.7    0.16       0
Bank Sta=4991.8,5010.4
Exp/Cntr=0.3,0.1

Type RM Length L Ch R = 1,260000,500,500,500
BEGIN DESCRIPTION:
Sweetwater Creek 518.0
END DESCRIPTION:
XS GIS Cut Line= 5
      1370219.64      6829409.32      1372207.13      6829444.56
      1372605.00      6829388.00      1372998.12      6829493.24
      1373284.40      6829482.79
#Sta/Elev= 30
  3012.2 2246.85  3157.6 2231.97  3637.7 2210.06  3687.7 2210.24  3717.7 2216.49
  3757.7 2204.99  4044.0 2207.61  4192.3 2209.76  4644.3 2206.82  4877.9 2209.37
  4947.9 2205.90  4987.9 2200.45  4992.8 2187.44  4993.3 2186.44  5011.4 2187.44
  5028.2 2190.20  5068.6 2204.86  5419.3 2215.80  5500.9 2215.28  5557.2 2215.77
  5571.9 2212.02  5588.2 2204.43  5602.6 2207.23  5619.5 2216.94  5681.4 2221.07
  5722.8 2227.76  5764.1 2239.29  5774.5 2247.68  5813.0 2255.55  6095.3 2266.40
#Mann=9,-1,0
  3012.2    0.07       0  4044.0   0.035       0  4192.3    0.07       0
  4644.3    0.16       0  4992.8    0.07       0  5011.4    0.16       0
  5500.9    0.07       0  5571.9    0.16       0  5602.6    0.07       0
Bank Sta=4992.8,5011.4
Exp/Cntr=0.3,0.1

Type RM Length L Ch R = 1,259500,562,562,562
BEGIN DESCRIPTION:
Sweetwater Creek 517.0
END DESCRIPTION:
XS GIS Cut Line= 3
      1370166.26      6829857.06      1372124.81      6829918.14
      1372931.13      6829982.67
#Sta/Elev= 30
  3040.5 2253.76  3209.3 2248.39  3269.4 2231.05  3299.4 2225.85  3459.4 2215.52
  3689.6 2206.95  3819.6 2205.03  3849.6 2211.58  3859.6 2210.32  3868.7 2204.14
  3889.7 2201.79  3919.7 2204.24  4820.7 2205.15  4940.2 2205.38  4990.2 2194.20
  4993.8 2187.78  4994.2 2186.78  5012.4 2187.78  5049.8 2198.04  5080.4 2202.19
  5228.0 2205.07  5291.1 2204.24  5321.2 2197.47  5351.3 2203.62  5561.8 2218.47
  5602.1 2223.48  5632.2 2231.69  5672.3 2246.54  5692.5 2258.73  5808.9 2261.84
#Mann=7,-1,0
  3040.5    0.07       0  4820.7    0.16       0  4993.8    0.07       0
  5012.4    0.16       0  5049.8    0.07       0  5228.0    0.16       0
  5561.8    0.07       0
Bank Sta=4993.8,5012.4
Exp/Cntr=0.3,0.1

Type RM Length L Ch R = 1,258938,438,438,438
BEGIN DESCRIPTION:
Sweetwater Creek 516.0
END DESCRIPTION:
XS GIS Cut Line= 4
      1370313.65      6830441.35      1372425.50      6830357.80
      1372730.90      6830303.34      1372936.05      6830195.69
#Sta/Elev= 30
  2886.5 2247.61  2927.9 2241.03  2967.9 2228.95  3068.0 2219.46  3258.1 2208.56
  3438.3 2202.14  3578.4 2201.33  3608.6 2206.96  3628.4 2200.43  3648.4 2198.21
  3678.5 2200.70  4367.8 2201.21  4519.1 2204.60  4719.3 2204.43  4839.4 2199.18
  4899.4 2199.58  4969.5 2193.90  4993.2 2186.14  4993.5 2185.14  5005.6 2186.14
  5009.6 2190.01  5019.8 2194.11  5070.6 2204.00  5182.3 2210.42  5298.5 2221.26
  5326.1 2224.06  5370.6 2232.92  5405.2 2252.25  5436.8 2260.43  5541.9 2266.46
#Mann=5,-1,0
  2886.5    0.07       0  4367.8    0.16       0  4993.2    0.07       0
  5005.6    0.16       0  5298.5    0.07       0
Bank Sta=4993.2,5005.6
Exp/Cntr=0.3,0.1

Type RM Length L Ch R = 1,258500,500,500,500
BEGIN DESCRIPTION:
Sweetwater Creek 515.0
END DESCRIPTION:
XS GIS Cut Line= 4
      1370312.82      6830698.48      1372309.61      6830738.79
      1372423.56      6830715.21      1373261.00      6830657.28
#Sta/Elev= 30
  3002.8 2251.96  3095.0 2244.43  3165.0 2225.00  3195.0 2222.97  3215.0 2217.80
  3515.1 2201.34  3695.1 2199.54  3735.1 2204.59  3765.1 2196.86  3795.1 2199.51
  4295.2 2198.38  4817.2 2203.25  4915.4 2203.55  4945.4 2200.52  4985.4 2192.82
  4994.9 2182.98  4995.2 2181.98  5007.3 2182.98  5024.7 2191.49  5074.9 2194.67
  5080.0 2190.93  5127.8 2200.17  5332.3 2208.74  5578.5 2215.95  5752.5 2229.37
  5849.5 2238.90  5868.8 2242.42  5879.6 2249.15  5899.7 2254.58  5955.8 2254.74
#Mann=6,-1,0
  3002.8    0.07       0  4817.2    0.16       0  4994.9    0.07       0
  5007.3    0.16       0  5332.3    0.07       0  5752.5    0.16       0
Bank Sta=4994.9,5007.3
Exp/Cntr=0.3,0.1

Type RM Length L Ch R = 1,258000,500,500,500
BEGIN DESCRIPTION:
Sweetwater Creek 514.0
END DESCRIPTION:
XS GIS Cut Line= 3
      1370289.05      6831018.43      1372149.25      6831190.09
      1373371.77      6831216.17
#Sta/Elev= 30
  3131.9 2254.05  3233.8 2245.18  3311.5 2227.41  3439.1 2213.43  3640.0 2201.78
  3830.2 2198.05  3850.9 2202.57  3891.1 2196.25  4050.3 2198.47  4291.4 2196.53
  4408.3 2195.16  4875.2 2201.90  4975.6 2191.23  4989.3 2179.95  4989.7 2178.95
  5007.9 2179.95  5015.8 2191.23  5065.8 2197.28  5346.6 2204.70  5615.9 2211.25
  5645.9 2217.27  5675.9 2213.06  5728.8 2214.88  5827.8 2219.97  6016.0 2234.76
  6066.0 2245.25  6082.5 2253.80  6093.1 2258.99  6126.0 2264.99  6222.8 2251.90
#Mann=13,-1,0
  3131.9    0.07       0  3233.8    0.16       0  3311.5    0.07       0
  4050.3    0.16       0  4291.4    0.07       0  4408.3    0.16       0
  4989.3    0.07       0  5007.9    0.16       0  5346.6    0.07       0
  5728.8    0.16       0  5827.8    0.07       0  6082.5    0.16       0
  6093.1    0.07       0
Bank Sta=4989.3,5007.9
Exp/Cntr=0.3,0.1

Type RM Length L Ch R = 1,257500,500,500,500
BEGIN DESCRIPTION:
Sweetwater Creek 513.0
END DESCRIPTION:
XS GIS Cut Line= 4
      1370313.38      6831381.62      1371613.22      6831601.81
      1371968.39      6831625.31      1373326.06      6831513.18
#Sta/Elev= 30
  3325.7 2251.37  3479.5 2245.45  3509.2 2231.96  3514.3 2233.79  3550.5 2221.89
  3629.9 2211.22  3854.8 2198.88  3976.5 2200.66  4006.9 2192.99  4112.5 2196.69
  4433.3 2194.36  4475.0 2187.59  4503.9 2192.71  4759.8 2196.43  4936.5 2199.57
  4975.7 2192.73  4986.6 2191.15  4995.7 2181.36  4996.1 2180.36  5014.3 2181.36
  5076.9 2192.97  5137.1 2197.13  5618.7 2204.23  6043.4 2227.58  6123.5 2235.06
  6170.6 2252.21  6206.5 2247.97  6260.9 2242.10  6331.1 2262.83  6362.3 2264.64
#Mann=9,-1,0
  3325.7    0.07       0  4112.5    0.16       0  4433.3    0.07       0
  4759.8    0.16       0  4975.7    0.07       0  4995.7    0.07       0
  5014.3    0.07       0  6043.4    0.16       0  6206.5    0.07       0
Bank Sta=4995.7,5014.3
Exp/Cntr=0.3,0.1

Type RM Length L Ch R = 1,257000,500,500,500
BEGIN DESCRIPTION:
Sweetwater Creek 512.0
END DESCRIPTION:
XS GIS Cut Line= 3
      1370413.95      6831577.09      1371904.59      6832068.67
      1372869.86      6832002.99
#Sta/Elev= 30
  3430.4 2249.66  3557.9 2247.67  3575.3 2239.12  3580.6 2243.28  3600.0 2224.78
  3638.8 2213.80  3821.1 2200.44  3936.9 2196.52  3961.7 2200.22  3993.5 2194.30
  4501.6 2193.28  4558.2 2185.78  4705.6 2193.38  4968.8 2194.25  4978.0 2193.78
  4989.9 2185.74  4993.8 2178.35  4994.3 2177.35  5012.5 2178.35  5030.5 2186.87
  5060.5 2184.05  5261.0 2199.03  5531.6 2200.94  5674.8 2207.97  5732.1 2217.12
  5772.2 2219.08  5823.7 2237.79  5842.4 2250.78  5852.4 2261.67  5967.5 2267.71
#Mann=3,-1,0
  3430.4    0.07       0  4993.8    0.07       0  5012.5    0.07       0
Bank Sta=4993.8,5012.5
Exp/Cntr=0.3,0.1

Type RM Length L Ch R = 1,256500,500,500,500
BEGIN DESCRIPTION:
Sweetwater Creek 511.0
END DESCRIPTION:
XS GIS Cut Line= 4
      1370505.02      6831738.01      1371504.15      6832269.72
      1371549.35      6832322.73      1372850.61      6832295.94
#Sta/Elev= 30
  3868.2 2252.67  3898.3 2248.87  3920.3 2234.91  3936.1 2230.05  3942.2 2223.99
  4015.4 2209.90  4260.5 2197.60  4304.4 2200.47  4332.6 2196.73  4500.5 2197.66
  4615.8 2199.45  4946.6 2194.15  4978.3 2184.54  4987.8 2177.88  4988.2 2176.88
  5006.5 2177.88  5006.7 2180.25  5013.2 2183.29  5069.7 2184.46  5105.3 2192.34
  5185.3 2192.50  5235.4 2182.89  5275.4 2192.26  5725.5 2197.80  6085.5 2209.81
  6165.5 2217.05  6225.6 2217.43  6303.5 2222.99  6335.6 2225.05  6371.2 2227.31
#Mann=6,-1,0
  3868.2    0.07       0  4500.5    0.16       0  4987.8    0.07       0
  5006.5    0.16       0  6303.5    0.16       0  6335.6    0.07       0
Bank Sta=4987.8,5006.5
Exp/Cntr=0.3,0.1

Type RM Length L Ch R = 1,256000,485,485,485
BEGIN DESCRIPTION:
Sweetwater Creek 510.0
END DESCRIPTION:
XS GIS Cut Line= 3
      1370364.78      6832736.51      1371478.09      6832711.00
      1373075.16      6832489.21
#Sta/Elev= 30
  3886.4 2219.18  3996.7 2214.56  4035.6 2203.36  4040.6 2204.56  4066.7 2198.05
  4216.7 2198.39  4326.7 2195.05  4791.4 2192.42  4896.9 2193.63  4917.3 2190.86
  4926.9 2187.57  4941.8 2186.89  4976.9 2186.15  4986.9 2183.63  4992.7 2177.39
  4993.1 2176.39  5011.5 2177.39  5017.1 2180.13  5037.3 2181.81  5055.3 2186.25
  5127.0 2190.25  5269.5 2193.16  5653.1 2194.19  5804.6 2199.62  5824.8 2202.30
  5859.0 2200.47  6107.4 2213.51  6145.7 2218.36  6294.1 2220.66  6612.4 2237.69
#Mann=5,-1,0
  3886.4    0.07       0  4791.4    0.16       0  4941.8    0.07       0
  4992.7    0.07       0  5011.5    0.07       0
Bank Sta=4992.7,5011.5
Exp/Cntr=0.3,0.1

Type RM Length L Ch R = 1,255515,515,515,515
BEGIN DESCRIPTION:
Sweetwater Creek 509.0
END DESCRIPTION:
XS GIS Cut Line= 3
      1370350.90      6832939.36      1371600.51      6833117.37
      1372991.87      6833093.33
#Sta/Elev= 30
  3732.9 2235.55  3760.5 2232.59  3848.2 2196.10  3925.8 2194.80  3999.8 2194.47
  4090.6 2193.13  4171.4 2195.50  4544.9 2190.79  4797.6 2192.22  4817.6 2191.69
  4838.0 2186.77  4899.3 2184.86  4964.2 2183.33  4987.4 2173.30  4987.9 2172.30
  5006.3 2173.30  5009.6 2179.40  5059.6 2192.51  5409.7 2189.10  5669.7 2197.34
  5709.7 2202.55  5719.7 2199.64  5739.7 2199.34  5789.7 2205.61  5959.8 2212.69
  6009.8 2218.62  6029.8 2215.88  6109.8 2223.81  6149.8 2224.42  6386.7 2239.43
#Mann=7,-1,0
  3732.9    0.07       0  3925.8    0.16       0  3999.8    0.07       0
  4544.9    0.16       0  4899.3    0.07       0  4987.4    0.07       0
  5006.3    0.07       0
Bank Sta=4987.4,5006.3
Exp/Cntr=0.3,0.1

Type RM Length L Ch R = 1,255000,500,500,500
BEGIN DESCRIPTION:
Sweetwater Creek 508.0
END DESCRIPTION:
XS GIS Cut Line= 3
      1370185.26      6833274.89      1371504.94      6833595.19
      1372454.99      6833938.00
#Sta/Elev= 30
  3642.0 2236.28  3671.9 2236.12  3718.8 2231.89  3754.9 2225.55  3772.3 2219.53
  3844.2 2199.02  3873.5 2196.66  3981.3 2190.58  4135.7 2189.58  4176.8 2192.09
  4197.4 2186.10  4225.3 2189.11  4454.7 2187.31  4523.6 2189.88  4653.4 2187.66
  4928.0 2189.32  4969.2 2183.80  4979.5 2179.62  4986.9 2171.88  4987.3 2170.88
  5005.7 2171.88  5019.5 2181.74  5024.8 2178.61  5063.8 2188.61  5090.0 2190.19
  5276.5 2186.72  5808.0 2188.32  5871.8 2193.03  5933.3 2209.73  6010.0 2211.54
#Mann=7,-1,0
  3642.0    0.07       0  3772.3    0.16       0  3873.5    0.07       0
  4523.6    0.16       0  4986.9    0.07       0  5005.7    0.16       0
  5090.0    0.07       0
Bank Sta=4986.9,5005.7
Exp/Cntr=0.3,0.1

Type RM Length L Ch R = 1,254500,500,500,500
BEGIN DESCRIPTION:
Sweetwater Creek 507.0
END DESCRIPTION:
XS GIS Cut Line= 3
      1370404.98      6833787.99      1371385.21      6834057.46
      1372354.95      6834237.99
#Sta/Elev= 30
  3983.4 2216.48  4000.6 2208.63  4005.8 2209.33  4045.6 2195.34  4074.7 2189.66
  4159.7 2189.17  4180.5 2186.39  4222.0 2189.81  4253.1 2185.39  4267.5 2187.00
  4584.4 2185.68  4699.0 2187.29  4796.0 2184.15  4885.7 2185.19  4958.3 2181.21
  4978.5 2181.86  4983.7 2180.87  4989.4 2176.05  4989.7 2170.02  4990.2 2169.02
  5008.6 2170.02  5020.1 2178.68  5027.7 2181.44  5050.6 2186.52  5085.6 2188.63
  5335.5 2184.87  5874.6 2187.03  5925.4 2191.24  5966.1 2203.50  5986.4 2205.02
#Mann=5,-1,0
  3983.4    0.07       0  4584.4    0.16       0  4796.0    0.07       0
  4989.7    0.07       0  5008.6    0.07       0
Bank Sta=4989.7,5008.6
Exp/Cntr=0.3,0.1

Type RM Length L Ch R = 1,254000,500,500,500
BEGIN DESCRIPTION:
Sweetwater Creek 506.0
END DESCRIPTION:
XS GIS Cut Line= 3
      1370505.03      6834138.01      1371027.30      6834315.19
      1372545.64      6834369.06
#Sta/Elev= 30
  4448.5 2190.79  4501.3 2187.28  4589.8 2188.17  4621.2 2185.72  4778.2 2183.01
  4903.8 2184.62  4944.8 2186.48  4955.3 2185.82  4961.3 2183.05  4976.5 2168.74
  4983.5 2168.74  4984.0 2167.74  5002.4 2168.74  5007.7 2181.80  5017.7 2181.68
  5037.7 2177.86  5077.8 2178.84  5097.8 2177.19  5107.8 2178.89  5197.8 2180.74
  5221.5 2182.96  5297.9 2185.98  5387.9 2187.80  5578.1 2184.11  6168.4 2188.51
  6238.5 2190.93  6268.5 2193.56  6338.5 2195.71  6388.6 2195.47  6519.3 2200.15
#Mann=3,-1,0
  4448.5    0.07       0  4983.5    0.07       0  5002.4    0.07       0
Bank Sta=4983.5,5002.4
Exp/Cntr=0.3,0.1

Type RM Length L Ch R = 1,253500,500,500,500
BEGIN DESCRIPTION:
Sweetwater Creek 505.0
END DESCRIPTION:
XS GIS Cut Line= 6
      1370177.76      6834303.59      1371206.45      6834658.69
      1371331.00      6834587.73      1371352.82      6834499.79
      1371833.98      6834496.44      1372466.28      6834609.48
#Sta/Elev= 30
  3768.4 2206.33  3934.7 2195.20  4114.6 2188.01  4137.7 2183.92  4168.9 2186.59
  4220.4 2185.78  4231.3 2183.40  4376.6 2182.20  4675.3 2186.28  4802.2 2181.70
  4858.7 2181.38  4891.8 2177.41  4929.3 2175.65  4945.1 2177.31  4950.9 2173.35
  4958.6 2174.62  4966.7 2171.99  4970.5 2165.73  4971.3 2164.73  5002.0 2165.73
  5002.4 2168.03  5030.6 2176.62  5036.6 2181.75  5083.1 2185.72  5152.8 2184.62
  5182.8 2186.04  5202.8 2184.25  5262.8 2183.66  5442.8 2184.46  6214.1 2194.37
#Mann=3,-1,0
  3768.4    0.07       0  4970.5    0.07       0  5002.0    0.07       0
Bank Sta=4970.5,5002
Exp/Cntr=0.3,0.1

Type RM Length L Ch R = 1,253000,500,500,500
BEGIN DESCRIPTION:
Sweetwater Creek 504.0
END DESCRIPTION:
XS GIS Cut Line= 3
      1370254.99      6834438.00      1371255.49      6834987.16
      1372205.04      6835338.01
#Sta/Elev= 30
  3858.7 2201.59  3984.2 2194.62  3991.8 2192.32  4035.4 2193.04  4100.8 2190.54
  4122.6 2188.55  4132.5 2185.78  4138.7 2180.73  4154.8 2184.30  4176.6 2185.80
  4258.0 2181.79  4807.8 2184.29  4911.1 2180.14  4976.6 2180.29  4996.9 2177.61
  5000.0 2164.70  5000.6 2163.70  5025.2 2164.70  5052.8 2175.27  5095.4 2178.51
  5102.1 2181.57  5114.5 2183.37  5416.7 2179.93  5663.6 2180.71  5708.9 2180.39
  5825.0 2185.79  5927.0 2192.55  5959.0 2199.08  5997.0 2210.03  6012.3 2211.51
#Mann=7,-1,0
  3858.7    0.07       0  5000.0    0.07       0  5025.2    0.07       0
  5114.5    0.16       0  5416.7    0.07       0  5663.6    0.16       0
  5825.0    0.07       0
Bank Sta=5000,5025.2
Exp/Cntr=0.3,0.1

Type RM Length L Ch R = 1,252500,500,500,500
BEGIN DESCRIPTION:
Sweetwater Creek 503.0
END DESCRIPTION:
XS GIS Cut Line= 3
      1369904.99      6834438.00      1370908.04      6835140.88
      1372804.98      6835987.99
#Sta/Elev= 30
  3775.2 2249.74  3797.4 2245.89  3854.1 2251.05  3897.3 2227.83  3940.4 2216.01
  4113.0 2198.83  4471.2 2179.56  4507.9 2183.87  4535.8 2179.63  4705.1 2181.60
  4870.0 2179.69  4982.1 2181.30  5003.7 2176.47  5009.2 2168.51  5009.3 2163.27
  5010.1 2162.27  5040.8 2163.27  5073.3 2163.61  5078.8 2173.03  5084.3 2173.81
  5095.2 2168.61  5107.5 2173.84  5281.4 2182.66  5790.3 2177.28  5813.5 2182.91
  6038.9 2178.09  6409.5 2188.01  6520.4 2197.31  6790.0 2209.76  7077.5 2218.63
#Mann=7,-1,0
  3775.2    0.07       0  4705.1    0.16       0  4870.0    0.07       0
  5009.3    0.07       0  5040.8    0.07       0  6520.4   0.035       0
  6790.0    0.07       0
Bank Sta=5009.3,5040.8
Exp/Cntr=0.3,0.1

Type RM Length L Ch R = 1,252000,500,500,500
BEGIN DESCRIPTION:
Sweetwater Creek 502.0
END DESCRIPTION:
XS GIS Cut Line= 4
      1369905.00      6834488.00      1370422.47      6835384.78
      1370610.49      6835489.93      1372361.14      6835904.62
#Sta/Elev= 30
  3749.2 2256.49  3772.3 2256.67  3784.4 2254.83  3797.6 2249.31  3816.0 2235.73
  3864.8 2218.36  3945.5 2208.38  4148.1 2194.03  4341.6 2182.86  4716.4 2177.82
  4722.2 2175.54  4797.3 2181.26  4824.7 2173.43  4862.4 2178.34  4889.8 2178.40
  4965.2 2175.37  4986.9 2169.85  4993.7 2166.23  4994.0 2162.35  4994.5 2161.35
  5012.9 2162.35  5045.7 2172.03  5066.3 2175.20  5136.2 2179.61  6073.4 2174.41
  6196.7 2175.60  6399.4 2179.76  6441.6 2183.60  6489.0 2181.91  6799.1 2202.08
#Mann=7,-1,0
  3749.2    0.07       0  3797.6    0.16       0  4148.1    0.07       0
  4889.8    0.16       0  4994.0    0.07       0  5012.9    0.16       0
  5136.2    0.07       0
Bank Sta=4994,5012.9
Exp/Cntr=0.3,0.1

Type RM Length L Ch R = 1,251500,500,500,500
BEGIN DESCRIPTION:
Sweetwater Creek 501.0
END DESCRIPTION:
XS GIS Cut Line= 3
      1369704.96      6836288.01      1370704.55      6835958.81
      1372361.88      6835982.76
#Sta/Elev= 30
  3947.6 2205.50  4053.7 2203.56  4179.3 2199.76  4242.4 2178.27  4313.3 2176.30
  4337.2 2174.03  4368.8 2178.48  4479.9 2176.76  4567.3 2174.00  4606.8 2178.09
  4621.5 2179.29  4653.0 2173.73  4718.0 2175.56  4916.2 2176.60  4979.4 2172.06
  4987.8 2161.24  4988.3 2160.24  5006.8 2161.24  5060.5 2166.63  5090.5 2173.38
  5220.5 2177.22  5760.5 2177.34  5790.5 2174.53  6020.6 2173.61  6217.2 2177.98
  6238.9 2177.75  6330.6 2180.13  6370.6 2185.18  6390.6 2181.70  6657.5 2201.58
#Mann=10,-1,0
  3947.6   0.035       0  4053.7    0.07       0  4313.3    0.12       0
  4479.9    0.07       0  4606.8    0.16       0  4718.0    0.07       0
  4987.8    0.07       0  5006.8    0.07       0  6217.2   0.035       0
  6238.9    0.07       0
Bank Sta=4987.8,5006.8
Exp/Cntr=0.3,0.1

Type RM Length L Ch R = 1,251000,458,458,458
BEGIN DESCRIPTION:
Sweetwater Creek 500.0
END DESCRIPTION:
XS GIS Cut Line= 3
      1369854.99      6836288.00      1370871.26      6836372.85
      1372755.03      6836038.00
#Sta/Elev= 30
  3980.2 2202.49  4020.3 2200.79  4037.9 2195.24  4042.9 2199.35  4080.6 2187.89
  4252.2 2178.18  4268.4 2177.30  4283.5 2176.96  4311.4 2168.95  4351.7 2175.54
  4391.6 2168.87  4431.8 2179.30  4450.8 2173.45  4626.6 2174.88  4853.2 2174.70
  4994.7 2159.51  4995.2 2158.51  5013.7 2159.51  5044.4 2170.73  5064.7 2170.93
  5074.9 2176.72  5085.1 2177.23  5775.7 2172.51  6167.0 2178.04  6257.2 2185.33
  6283.6 2183.01  6364.8 2188.03  6433.2 2194.76  6660.3 2209.93  6913.3 2218.45
#Mann=10,-1,0
  3980.2    0.07       0  4252.2    0.12       0  4268.4   0.035       0
  4351.7    0.07       0  4450.8   0.035       0  4626.6    0.07       0
  4994.7    0.07       0  5013.7    0.07       0  6167.0   0.035       0
  6433.2    0.07       0
Bank Sta=4994.7,5013.7
Exp/Cntr=0.3,0.1

Type RM Length L Ch R = 1,250542,542,542,542
BEGIN DESCRIPTION:
Sweetwater Creek 499.0
END DESCRIPTION:
XS GIS Cut Line= 4
      1370104.99      6836538.00      1370416.64      6836501.77
      1370639.68      6836648.30      1372220.37      6836203.50
#Sta/Elev= 30
  4596.1 2203.67  4611.2 2200.94  4656.5 2183.89  4811.2 2163.00  4827.7 2162.42
  4857.9 2172.13  4935.9 2174.76  4955.8 2174.47  4964.2 2171.31  4979.3 2170.92
  4991.6 2166.48  4992.4 2159.21  4992.9 2158.21  5011.4 2159.21  5027.5 2161.28
  5057.6 2159.93  5072.7 2161.42  5099.8 2170.00  5143.9 2171.84  5231.1 2175.46
  5298.7 2175.75  5485.2 2175.67  6160.0 2171.18  6480.8 2174.11  6653.3 2179.12
  6699.0 2180.84  6719.7 2185.98  6746.3 2183.49  6787.5 2187.36  6818.8 2190.28
#Mann=11,-1,0
  4596.1   0.035       0  4611.2    0.07       0  4811.2   0.035       0
  4935.9    0.07       0  4992.4    0.07       0  5011.4    0.07       0
  5143.9    0.07       0  5298.7    0.16       0  5485.2    0.07       0
  6653.3   0.035       0  6787.5    0.07       0
Bank Sta=4992.4,5011.4
Exp/Cntr=0.3,0.1

Type RM Length L Ch R = 1,250000,425,425,425
BEGIN DESCRIPTION:
Sweetwater Creek 498.0
END DESCRIPTION:
XS GIS Cut Line= 3
      1370154.95      6836938.00      1370483.66      6836967.19
      1372404.97      6836188.01
#Sta/Elev= 30
  4670.0 2212.51  4710.2 2206.40  4725.0 2199.88  4730.9 2199.87  4750.4 2179.72
  4790.5 2176.22  4810.6 2178.11  4842.7 2173.39  4896.3 2173.13  4941.1 2169.88
  4949.4 2165.46  4954.4 2168.99  4961.2 2162.65  4979.9 2158.11  4980.5 2157.11
  5005.2 2158.11  5086.7 2160.30  5109.4 2163.38  5129.8 2170.85  5144.9 2172.94
  5237.9 2174.16  5519.4 2173.17  6188.5 2170.44  6544.6 2174.02  6688.9 2178.01
  6760.4 2181.64  6782.0 2185.54  6820.1 2184.32  6897.8 2192.15  7073.3 2203.66
#Mann=9,-1,0
  4670.0   0.035       0  4725.0    0.07       0  4896.3   0.035       0
  4979.9   0.035       0  5005.2   0.035       0  5129.8    0.07       0
  5144.9   0.035       0  5237.9    0.16       0  5519.4    0.07       0
Bank Sta=4979.9,5005.2
Exp/Cntr=0.3,0.1

Type RM Length L Ch R = 1,249575,575,575,575
BEGIN DESCRIPTION:
Sweetwater Creek 497.0
END DESCRIPTION:
XS GIS Cut Line= 5
      1370254.98      6837187.99      1370471.04      6837306.21
      1370654.50      6837322.80      1370868.31      6837291.65
      1372298.40      6836322.34
#Sta/Elev= 30
  4569.5 2176.13  4583.3 2177.71  4619.1 2169.89  4681.0 2171.49  4730.2 2169.24
  4752.1 2168.81  4774.7 2157.71  4790.0 2156.18  4820.3 2162.58  4991.6 2154.52
  4992.2 2153.52  5016.9 2154.52  5030.8 2160.29  5121.8 2156.35  5131.9 2158.43
  5142.2 2170.02  5152.1 2170.65  5266.8 2168.91  5302.7 2171.48  5440.5 2167.38
  5554.3 2170.27  5770.0 2171.37  6159.3 2169.49  6324.1 2170.71  6647.7 2177.57
  6764.4 2182.29  6779.3 2186.38  6800.3 2184.09  6829.3 2186.49  6943.7 2193.36
#Mann=7,-1,0
  4569.5    0.07       0  4619.1   0.035       0  4730.2    0.07       0
  4991.6    0.07       0  5016.9    0.07       0  6647.7   0.035       0
  6829.3    0.07       0
Bank Sta=4991.6,5016.9
Exp/Cntr=0.3,0.1

Type RM Length L Ch R = 1,249000,500,500,500
BEGIN DESCRIPTION:
Sweetwater Creek 496.0
END DESCRIPTION:
XS GIS Cut Line= 4
      1370499.50      6838365.14      1370609.19      6837733.70
      1370669.28      6837610.95      1372296.85      6836420.39
#Sta/Elev= 30
  4359.1 2175.91  4416.2 2177.38  4427.2 2171.72  4481.0 2168.76  4535.6 2171.27
  4540.6 2174.54  4579.5 2176.96  4595.2 2181.32  4649.8 2172.31  4654.9 2164.17
  4681.0 2165.80  4701.3 2174.18  4752.0 2179.93  4774.2 2173.06  4823.1 2170.80
  4853.5 2163.27  4991.9 2154.26  4992.4 2153.26  5012.2 2154.26  5135.5 2159.16
  5151.7 2166.20  5179.4 2171.37  5240.0 2170.78  5737.6 2167.01  5980.1 2170.95
  6366.9 2169.13  6947.0 2178.78  7017.0 2181.53  7039.4 2185.56  7153.2 2187.90
#Mann=6,-1,0
  4359.1    0.07       0  4991.9    0.07       0  5012.2    0.07       0
  5151.7    0.16       0  5240.0    0.07       0  6947.0   0.035       0
Bank Sta=4991.9,5012.2
Exp/Cntr=0.3,0.1

Type RM Length L Ch R = 1,248500,500,500,500
BEGIN DESCRIPTION:
Sweetwater Creek 495.0
END DESCRIPTION:
XS GIS Cut Line= 4
      1370694.85      6839161.56      1371033.64      6837709.15
      1371004.54      6837446.40      1372366.56      6836616.50
#Sta/Elev= 30
  3508.6 2178.48  3851.1 2167.83  4518.6 2169.72  4549.4 2156.43  4568.3 2154.77
  4591.7 2157.57  4600.7 2162.77  4634.2 2169.46  4739.0 2170.14  4766.6 2170.56
  4888.2 2170.51  4894.6 2163.57  4899.8 2166.40  4919.0 2152.93  4954.3 2150.50
  4955.0 2149.50  4988.1 2150.50  4990.9 2153.56  5034.7 2155.99  5071.6 2171.15
  5101.8 2169.90  5120.4 2165.68  5181.1 2169.05  5381.2 2170.26  5497.4 2166.37
  5745.0 2170.27  6210.1 2169.40  6778.3 2183.79  6842.2 2187.04  6859.3 2188.73
#Mann=9,-1,0
  3508.6    0.07       0  4568.3    0.16       0  4739.0    0.07       0
  4766.6    0.16       0  4954.3    0.07       0  4988.1    0.16       0
  5181.1    0.07       0  6778.3   0.035       0  6842.2    0.07       0
Bank Sta=4954.3,4988.1
Exp/Cntr=0.3,0.1

Type RM Length L Ch R = 1,248000,500,500,500
BEGIN DESCRIPTION:
Sweetwater Creek 494.0
END DESCRIPTION:
XS GIS Cut Line= 4
      1370847.58      6839319.80      1371338.53      6837387.49
      1371377.75      6837242.49      1372550.36      6836810.68
#Sta/Elev= 30
  3006.3 2177.37  3070.1 2171.19  3224.8 2166.61  4091.5 2168.72  4109.8 2168.03
  4132.8 2158.07  4163.7 2154.34  4191.7 2158.10  4215.3 2168.04  4362.3 2169.54
  4462.6 2168.56  4700.3 2167.59  4741.5 2172.05  4751.8 2171.19  4759.7 2165.74
  4764.8 2169.52  4782.8 2157.06  4793.1 2155.16  4887.6 2156.15  4916.9 2152.66
  4978.8 2152.60  4992.7 2148.56  4993.0 2147.56  5006.2 2148.56  5039.8 2160.60
  5092.7 2169.92  5658.8 2169.38  5819.1 2174.37  5960.8 2174.50  6399.8 2190.50
#Mann=5,-1,0
  3006.3    0.07       0  4362.3   0.035       0  4462.6    0.07       0
  4992.7    0.07       0  5006.2    0.07       0
Bank Sta=4992.7,5006.2
Exp/Cntr=0.3,0.1

Type RM Length L Ch R = 1,247500,500,500,500
BEGIN DESCRIPTION:
Sweetwater Creek 493.0
END DESCRIPTION:
XS GIS Cut Line= 4
      1370857.53      6839381.97      1371398.62      6837896.65
      1371604.85      6837747.20      1372579.46      6836972.98
#Sta/Elev= 30
  3164.5 2178.81  3221.9 2179.61  3264.6 2171.38  3351.0 2167.00  4286.7 2167.93
  4328.8 2167.17  4342.5 2159.46  4367.8 2154.25  4392.7 2156.09  4403.7 2160.58
  4417.8 2162.34  4428.9 2167.26  4435.2 2167.58  4624.2 2167.70  4676.4 2168.34
  4801.9 2168.80  4885.4 2165.74  4906.2 2162.21  4927.1 2153.88  4992.1 2149.35
  4992.6 2146.48  4992.9 2145.48  5006.2 2146.48  5006.7 2149.49  5027.5 2152.22
  5041.9 2160.31  5085.2 2167.62  5689.8 2171.68  6174.6 2186.04  6244.7 2189.83
#Mann=7,-1,0
  3164.5    0.07       0  4417.8   0.035       0  4624.2    0.07       0
  4676.4   0.035       0  4801.9    0.07       0  4992.6    0.07       0
  5006.2    0.07       0
Bank Sta=4992.6,5006.2
Exp/Cntr=0.3,0.1

Type RM Length L Ch R = 1,247000,500,500,500
BEGIN DESCRIPTION:
Sweetwater Creek 492.0
END DESCRIPTION:
XS GIS Cut Line= 3
      1370928.03      6839380.64      1371899.21      6838132.34
      1372599.26      6837249.64
#Sta/Elev= 30
  3418.4 2175.33  3460.1 2167.65  3532.5 2165.69  4167.1 2166.72  4424.6 2165.30
  4525.3 2164.84  4536.7 2162.60  4558.6 2151.91  4579.5 2148.83  4614.7 2150.06
  4629.2 2151.81  4637.4 2155.57  4643.7 2153.85  4664.5 2162.71  4672.7 2161.54
  4679.0 2165.42  4857.3 2166.69  4915.2 2162.30  4942.3 2150.13  4979.4 2149.98
  4989.7 2146.45  4990.2 2145.45  5010.1 2146.45  5043.5 2164.52  5056.6 2166.43
  5232.6 2166.12  5434.4 2167.44  5836.2 2177.79  6046.4 2181.38  6126.6 2183.51
#Mann=9,-1,0
  3418.4    0.07       0  4167.1    0.16       0  4424.6    0.07       0
  4525.3    0.16       0  4989.7    0.07       0  5010.1    0.16       0
  5232.6    0.07       0  5836.2   0.035       0  6046.4    0.07       0
Bank Sta=4989.7,5010.1
Exp/Cntr=0.3,0.1

Type RM Length L Ch R = 1,246500,500,500,500
BEGIN DESCRIPTION:
Sweetwater Creek 491.0
END DESCRIPTION:
XS GIS Cut Line= 3
      1370971.14      6839566.83      1372110.06      6838543.39
      1372766.58      6837713.72
#Sta/Elev= 30
  3468.8 2177.40  3491.8 2176.16  3513.5 2169.13  3548.6 2166.46  4262.8 2164.56
  4606.2 2163.31  4639.2 2162.61  4667.6 2157.01  4702.7 2155.95  4717.0 2153.33
  4755.5 2155.66  4802.2 2164.12  4929.2 2166.74  4950.9 2164.05  4965.1 2154.33
  4971.8 2153.60  4979.3 2148.35  4987.8 2145.62  4988.2 2144.62  5008.1 2145.62
  5014.6 2148.05  5057.9 2149.61  5064.3 2154.72  5070.7 2155.52  5078.7 2161.03
  5134.8 2164.37  5394.5 2164.24  5562.8 2164.77  5825.6 2170.04  6058.0 2178.17
#Mann=7,-1,0
  3468.8    0.07       0  4262.8    0.16       0  4606.2    0.07       0
  4755.5    0.16       0  4987.8    0.07       0  5008.1    0.16       0
  5394.5    0.07       0
Bank Sta=4987.8,5008.1
Exp/Cntr=0.3,0.1

Type RM Length L Ch R = 1,246000,611,611,611
BEGIN DESCRIPTION:
Sweetwater Creek 490.0
END DESCRIPTION:
XS GIS Cut Line= 3
      1371276.60      6839549.92      1372541.45      6838737.84
      1373147.80      6838156.95
#Sta/Elev= 30
  3496.9 2165.33  3851.7 2164.03  4388.6 2162.36  4489.0 2163.05  4510.1 2154.37
  4531.3 2151.56  4546.5 2145.27  4567.6 2146.77  4576.4 2149.44  4582.0 2153.41
  4625.1 2162.05  4661.4 2164.14  4879.4 2163.28  4952.1 2150.59  4967.3 2149.65
  4973.2 2146.97  4980.5 2148.95  4994.4 2148.74  4996.9 2144.01  4997.4 2143.01
  5017.3 2144.01  5037.7 2145.09  5051.9 2152.23  5059.1 2151.56  5080.2 2161.38
  5087.4 2162.74  5150.9 2159.88  5205.2 2160.17  5525.8 2169.33  5839.7 2183.29
#Mann=7,-1,0
  3496.9    0.07       0  3851.7    0.16       0  4388.6    0.07       0
  4582.0    0.16       0  4996.9    0.07       0  5017.3    0.16       0
  5205.2    0.07       0
Bank Sta=4996.9,5017.3
Exp/Cntr=0.3,0.1

Type RM Length L Ch R = 1,245389,389,389,389
BEGIN DESCRIPTION:
Sweetwater Creek 489.0
END DESCRIPTION:
XS GIS Cut Line= 3
      1371696.89      6839545.32      1372811.49      6839144.74
      1373154.98      6838838.02
#Sta/Elev= 30
  3815.6 2162.62  3862.7 2162.45  3941.9 2162.07  4214.2 2161.43  4227.0 2161.29
  4506.1 2160.58  4525.5 2154.23  4531.5 2148.89  4536.8 2149.26  4556.9 2143.76
  4592.9 2155.42  4610.6 2156.92  4618.3 2159.83  4623.6 2157.79  4685.1 2161.43
  4742.0 2161.37  4940.0 2161.98  4971.1 2159.21  4982.5 2149.42  4987.8 2140.58
  4988.2 2139.58  5008.1 2140.58  5042.9 2145.38  5057.1 2153.55  5071.4 2158.49
  5129.3 2160.72  5212.7 2160.10  5345.7 2163.27  5349.1 2163.38  5460.5 2166.76
#Mann=11,-1,0
  3815.6    0.07       0  3862.7    0.16       0  3941.9    0.07       0
  4214.2    0.16       0  4227.0    0.07       0  4742.0    0.16       0
  4987.8    0.07       0  5008.1    0.16       0  5129.3    0.07       0
  5345.7    0.16       0  5349.1    0.07       0
Bank Sta=4987.8,5008.1
Exp/Cntr=0.3,0.1

Type RM Length L Ch R = 1,245000,500,500,500
BEGIN DESCRIPTION:
Sweetwater Creek 488.0
END DESCRIPTION:
XS GIS Cut Line= 3
      1371889.04      6839882.68      1373058.31      6839434.83
      1373304.99      6839088.01
#Sta/Elev= 30
  3747.9 2164.43  3797.1 2161.58  3925.6 2160.08  4366.0 2159.49  4385.4 2157.24
  4390.7 2158.30  4415.4 2150.25  4420.8 2153.29  4445.5 2146.75  4450.8 2148.05
  4470.2 2145.80  4475.5 2147.52  4500.2 2147.92  4537.4 2158.30  4632.4 2157.71
  4754.5 2159.69  4771.6 2161.47  4900.1 2161.70  4964.3 2155.90  4973.4 2151.23
  4978.8 2146.27  4985.7 2143.88  4987.5 2140.66  4988.1 2139.66  5014.6 2140.66
  5045.2 2145.42  5066.9 2156.76  5082.0 2159.61  5189.5 2158.82  5425.6 2164.26
#Mann=5,-1,0
  3747.9    0.07       0  4537.4    0.16       0  4987.5    0.07       0
  5014.6    0.16       0  5066.9    0.07       0
Bank Sta=4987.5,5014.6
Exp/Cntr=0.3,0.1

Type RM Length L Ch R = 1,244500,500,500,500
BEGIN DESCRIPTION:
Sweetwater Creek 487.0
END DESCRIPTION:
XS GIS Cut Line= 3
      1372286.40      6840166.29      1373487.76      6839588.22
      1373604.99      6839388.02
#Sta/Elev= 30
  3666.8 2167.29  3700.8 2168.71  3731.8 2160.23  3754.0 2159.14  3911.0 2157.79
  4213.1 2155.99  4317.3 2155.62  4322.8 2149.77  4345.5 2144.87  4375.5 2142.15
  4411.8 2145.13  4430.4 2148.72  4436.0 2153.90  4481.2 2157.67  4741.7 2159.93
  4898.9 2155.81  4944.9 2141.85  4973.5 2138.55  4974.1 2137.55  5000.6 2138.55
  5002.2 2142.85  5020.9 2148.64  5048.2 2146.15  5056.7 2150.11  5063.9 2148.00
  5069.8 2151.63  5085.4 2150.68  5122.6 2159.05  5224.1 2163.59  5232.0 2164.03
#Mann=9,-1,0
  3666.8    0.07       0  3911.0    0.16       0  4213.1    0.07       0
  4411.8    0.16       0  4898.9    0.07       0  4973.5    0.07       0
  5000.6    0.07       0  5056.7    0.16       0  5224.1    0.07       0
Bank Sta=4973.5,5000.6
Exp/Cntr=0.3,0.1

Type RM Length L Ch R = 1,244000,500,500,500
BEGIN DESCRIPTION:
Sweetwater Creek 486.0
END DESCRIPTION:
XS GIS Cut Line= 3
      1372716.44      6840371.90      1373739.09      6839922.84
      1374155.01      6839437.99
#Sta/Elev= 30
  3883.1 2156.28  4222.2 2153.05  4296.5 2151.95  4581.4 2156.80  4591.4 2156.22
  4613.3 2146.82  4622.6 2146.77  4628.1 2142.86  4635.1 2142.68  4657.0 2145.34
  4721.5 2144.38  4727.0 2147.25  4733.4 2145.78  4750.3 2148.22  4755.8 2151.68
  4831.7 2158.13  4901.4 2158.57  4930.2 2152.26  4948.1 2144.05  4989.8 2134.32
  4990.2 2133.32  5010.1 2134.32  5021.4 2152.22  5029.1 2150.14  5035.7 2157.49
  5057.7 2151.97  5113.6 2156.74  5262.6 2162.70  5539.5 2180.86  5638.8 2189.93
#Mann=5,-1,0
  3883.1    0.07       0  4222.2    0.16       0  4989.8    0.07       0
  5010.1    0.16       0  5262.6    0.07       0
Bank Sta=4989.8,5010.1
Exp/Cntr=0.3,0.1

Type RM Length L Ch R = 1,243500,500,500,500
BEGIN DESCRIPTION:
Sweetwater Creek 485.0
END DESCRIPTION:
XS GIS Cut Line= 3
      1372389.52      6840874.61      1374012.06      6840288.37
      1374285.43      6839487.12
#Sta/Elev= 30
  3274.8 2155.53  3554.0 2154.27  3577.3 2154.35  3706.6 2154.17  3838.8 2153.51
  3886.7 2137.03  3918.6 2138.35  3961.4 2152.76  3971.8 2153.72  4265.5 2149.71
  4354.5 2148.62  4869.4 2157.89  4942.0 2156.03  4956.1 2152.85  4961.4 2144.37
  4981.5 2140.28  4983.4 2134.42  4984.0 2133.42  5010.6 2134.42  5011.0 2139.48
  5032.1 2142.49  5158.9 2146.00  5177.1 2153.79  5208.4 2156.19  5219.5 2162.58
  5232.8 2161.50  5239.7 2156.86  5264.5 2154.79  5400.6 2160.88  5846.6 2191.24
#Mann=10,-1,0
  3274.8    0.16       0  3554.0    0.07       0  3577.3    0.16       0
  3706.6    0.07       0  4265.5    0.16       0  4942.0    0.07       0
  4983.4    0.07       0  5010.6    0.07       0  5219.5    0.16       0
  5400.6    0.07       0
Bank Sta=4983.4,5010.6
Exp/Cntr=0.3,0.1

Type RM Length L Ch R = 1,243000,500,500,500
BEGIN DESCRIPTION:
Sweetwater Creek 484.0
END DESCRIPTION:
XS GIS Cut Line= 4
      1372377.44      6841346.40      1374310.46      6840564.84
      1374455.72      6840238.78      1374555.01      6840037.98
#Sta/Elev= 30
  2558.0 2161.31  2684.7 2149.21  2700.7 2140.64  2738.7 2150.73  2843.4 2150.31
  2992.4 2150.48  3100.0 2151.10  3524.1 2149.73  3583.2 2142.44  3607.3 2133.44
  3666.4 2152.28  3858.6 2148.97  3939.0 2146.36  4387.5 2152.76  4658.2 2153.81
  4736.4 2154.81  4753.8 2146.42  4771.0 2139.27  4817.1 2139.11  4834.8 2143.80
  4869.5 2166.51  4882.5 2162.96  4902.3 2154.57  5000.0 2139.98  5000.8 2133.43
  5001.4 2132.43  5028.0 2133.43  5073.5 2146.95  5223.3 2161.13  5224.0 2161.13
#Mann=15,-1,0
  2558.0    0.07       0  2684.7    0.16       0  2843.4    0.07       0
  2992.4    0.16       0  3100.0    0.07       0  3858.6    0.16       0
  3939.0    0.07       0  4387.5    0.16       0  4658.2    0.07       0
  4753.8    0.16       0  4882.5    0.07       0  5000.8    0.07       0
  5028.0    0.07       0  5073.5    0.16       0  5223.3    0.07       0
Bank Sta=5000.8,5028
Exp/Cntr=0.3,0.1

Type RM Length L Ch R = 1,242500,479,479,479
BEGIN DESCRIPTION:
Sweetwater Creek 483.0
END DESCRIPTION:
XS GIS Cut Line= 4
      1372444.30      6841388.47      1374662.01      6840580.20
      1374904.71      6840288.08      1374854.99      6840087.96
#Sta/Elev= 30
  2259.8 2160.33  2383.1 2150.34  2443.6 2142.89  2448.9 2140.10  2462.8 2149.38
  2590.5 2146.07  2666.0 2149.60  2754.1 2149.67  3155.9 2153.58  3197.2 2150.38
  3211.7 2143.93  3233.6 2124.06  3235.1 2123.06  3301.5 2124.06  3303.6 2137.60
  3314.3 2147.73  3346.2 2151.05  3367.5 2159.54  3384.5 2155.04  3654.8 2144.11
  3764.9 2149.37  3791.2 2149.68  4507.6 2152.50  4577.1 2153.67  4964.5 2149.44
  4993.1 2138.61  4996.8 2132.88  5010.4 2132.28  5123.7 2156.40  5206.2 2165.16
#Mann=11,-1,0
  2259.8    0.07       0  2383.1    0.16       0  2443.6    0.07       0
  2666.0    0.16       0  2754.1    0.07       0  3233.6    0.07       0
  3301.5    0.07       0  3764.9    0.16       0  3791.2    0.07       0
  4507.6    0.16       0  4577.1    0.07       0
Bank Sta=3233.6,3301.5
Exp/Cntr=0.3,0.1

Type RM Length L Ch R = 1,242021,1021,1021,1021
BEGIN DESCRIPTION:
Sweetwater Creek 482.0
END DESCRIPTION:
XS GIS Cut Line= 3
      1372478.32      6841444.13      1375351.16      6840412.90
      1375665.40      6840242.89
#Sta/Elev= 30
  1963.9 2162.44  2171.0 2150.14  2176.3 2143.18  2194.1 2139.82  2289.3 2141.29
  2293.9 2148.35  2495.4 2147.34  2826.0 2154.01  2882.1 2149.15  2887.4 2144.47
  2893.2 2123.94  2894.7 2122.94  2961.2 2123.94  2974.3 2124.70  3012.2 2149.50
  3161.0 2162.35  3184.2 2153.59  3373.5 2142.68  3558.6 2150.53  3667.0 2151.01
  4169.2 2152.45  4317.3 2152.27  4850.3 2150.61  5021.2 2134.89  5037.3 2135.86
  5053.5 2145.42  5059.2 2150.20  5066.1 2167.68  5075.4 2171.06  5373.5 2180.72
#Mann=9,-1,0
  1963.9    0.07       0  2289.3    0.16       0  2495.4    0.07       0
  2893.2    0.07       0  2961.2    0.07       0  3558.6    0.16       0
  3667.0    0.07       0  4169.2    0.16       0  4317.3    0.07       0
Bank Sta=2893.2,2961.2
Exp/Cntr=0.3,0.1

Type RM Length L Ch R = 1,241000,428,428,428
BEGIN DESCRIPTION:
Sweetwater Creek 480.0
END DESCRIPTION:
XS GIS Cut Line= 4
      1372439.61      6841535.75      1374794.33      6840962.74
      1375155.89      6841304.85      1375649.59      6841178.17
#Sta/Elev= 30
  2078.8 2178.24  2131.7 2171.37  2136.8 2167.42  2256.9 2154.90  2893.1 2146.78
  2898.3 2141.66  2934.9 2137.35  3060.1 2155.07  3134.1 2147.48  3143.5 2143.99
  3148.7 2134.45  3161.9 2121.97  3163.4 2120.97  3229.9 2121.97  3257.6 2129.23
  3279.0 2143.86  3288.5 2139.59  3315.6 2150.11  3336.7 2152.33  3628.1 2144.63
  3918.3 2149.27  4938.0 2151.19  4959.0 2148.12  4980.4 2136.70  5002.1 2131.10
  5071.4 2138.05  5102.3 2146.18  5133.3 2144.05  5236.5 2160.05  5509.7 2161.74
#Mann=5,-1,0
  2078.8    0.07       0  3161.9    0.07       0  3229.9    0.07       0
  3336.7    0.16       0  3918.3    0.07       0
Bank Sta=3161.9,3229.9
Exp/Cntr=0.3,0.1
