HEC-RAS study Chimney Creek.prj: Chimney Creek Base Level Engineering

--- Chimney Creek.g01 (geometry) --- (continued)

Type RM Length L Ch R = 1,38306,403,403,403
BEGIN DESCRIPTION:
Mapping XS c6a3fcbd
END DESCRIPTION:
XS GIS Cut Line= 3
      1645885.15      6950293.34      1645460.88      6951293.79
      1645458.07      6951918.38
#Sta/Elev= 30
  3919.5 1668.23  3946.3 1668.29  3978.7 1666.15  4189.8 1664.30  4348.2 1661.82
  4402.5 1660.19  4571.9 1661.87  4760.9 1661.03  4815.3 1659.51  4847.8 1656.01
  4869.6 1654.99  4891.3 1656.60  4954.1 1654.79  4977.8 1655.23  4981.4 1652.85
  4982.3 1652.35  5018.5 1652.85  5020.4 1654.93  5030.4 1658.29  5040.4 1659.97
  5050.4 1660.38  5080.4 1661.34  5320.4 1661.53  5380.4 1663.10  5400.4 1665.39
  5428.0 1666.83  5460.4 1669.34  5500.4 1670.73  5550.4 1674.06  5630.8 1677.82
#Mann=4,-1,0
  3919.5   0.035       0  4981.4   0.035       0  5018.5   0.035       0
  5428.0    0.07       0
Bank Sta=4981.4,5018.5
Exp/Cntr=0.3,0.1

Type RM Length L Ch R = 1,37903,537,537,537
BEGIN DESCRIPTION:
Mapping XS 437c863d
END DESCRIPTION:
XS GIS Cut Line= 3
      1644909.46      6950362.82      1645113.22      6951138.84
      1645318.71      6951774.53
#Sta/Elev= 30
  4199.0 1674.35  4204.3 1673.79  4240.5 1672.06  4256.0 1670.03  4287.1 1667.58
  4483.5 1662.59  4512.7 1660.16  4593.5 1656.62  4700.6 1655.13  4762.7 1658.08
  4835.7 1657.85  4928.1 1655.25  4946.4 1653.39  4992.0 1653.08  4992.4 1651.27
  4993.4 1650.77  5029.5 1651.27  5032.0 1653.06  5051.8 1657.46  5057.1 1656.72
  5063.5 1658.16  5083.8 1658.91  5190.4 1660.35  5494.4 1659.31  5568.0 1661.29
  5599.5 1663.55  5606.7 1664.83  5630.8 1665.67  5638.7 1667.17  5669.4 1668.54
#Mann=5,-1,0
  4199.0    0.07       0  4204.3   0.035       0  4992.4   0.035       0
  5029.5   0.035       0  5630.8    0.07       0
Bank Sta=4992.4,5029.5
Exp/Cntr=0.3,0.1

Type RM Length L Ch R = 1,37366,614,614,614
BEGIN DESCRIPTION:
Mapping XS a59f637a
END DESCRIPTION:
XS GIS Cut Line= 3
      1644402.01      6950750.03      1644612.05      6951046.87
      1645172.82      6951838.55
#Sta/Elev= 30
  4640.1 1677.98  4662.1 1677.49  4684.5 1675.62  4690.6 1674.02  4705.4 1673.80
  4711.6 1672.62  4806.4 1667.08  4848.2 1663.46  4883.9 1662.59  4944.7 1655.92
  4956.1 1654.13  4970.0 1648.65  4978.7 1646.54  4995.5 1646.10  4996.5 1645.60
  5033.2 1646.10  5041.9 1646.49  5071.0 1655.38  5078.6 1656.47  5100.5 1657.05
  5171.9 1656.91  5178.0 1657.61  5201.2 1656.99  5386.0 1658.94  5789.4 1658.17
  5861.0 1659.54  5896.7 1661.17  5911.2 1662.71  5953.3 1665.18  5973.9 1667.14
#Mann=5,-1,0
  4640.1    0.07       0  4944.7   0.035       0  4995.5   0.035       0
  5033.2   0.035       0  5911.2    0.07       0
Bank Sta=4995.5,5033.2
Exp/Cntr=0.3,0.1

Type RM Length L Ch R = 1,36752,391,391,391
BEGIN DESCRIPTION:
Mapping XS 91945e19
END DESCRIPTION:
XS GIS Cut Line= 3
      1644103.41      6951388.04      1644351.64      6951539.06
      1645050.65      6951938.00
#Sta/Elev= 30
  4711.0 1684.23  4748.0 1682.14  4762.3 1680.30  4777.7 1676.49  4793.2 1673.88
  4841.7 1668.17  4894.0 1658.72  4900.1 1655.71  4909.5 1652.98  4921.0 1650.90
  4936.6 1649.31  4967.6 1648.60  4970.0 1647.87  4971.0 1647.37  5007.8 1647.87
  5016.9 1648.89  5031.9 1647.89  5047.8 1651.10  5063.0 1650.21  5069.4 1651.34
  5097.5 1650.91  5112.6 1651.77  5128.4 1653.86  5150.0 1655.07  5193.2 1656.12
  5311.3 1657.30  5569.1 1656.67  5683.7 1657.74  5752.0 1660.60  5806.4 1665.84
#Mann=5,-1,0
  4711.0    0.07       0  4921.0   0.035       0  4970.0   0.035       0
  5007.8   0.035       0  5683.7    0.07       0
Bank Sta=4970,5007.8
Exp/Cntr=0.3,0.1

Type RM Length L Ch R = 1,36361,371,371,371
BEGIN DESCRIPTION:
Mapping XS 1970db4e
END DESCRIPTION:
XS GIS Cut Line= 3
      1643849.57      6951793.23      1644212.83      6951883.07
      1644962.62      6952123.47
#Sta/Elev= 30
  4626.1 1685.47  4734.7 1681.07  4775.9 1678.51  4786.2 1677.09  4791.6 1675.03
  4806.8 1671.35  4868.6 1664.06  4874.4 1662.47  4899.5 1658.98  4909.8 1656.70
  4915.8 1653.82  4930.4 1652.52  4938.2 1651.82  4971.6 1649.60  4992.2 1647.11
  4998.7 1645.10  5011.9 1644.59  5012.9 1644.09  5049.7 1644.59  5051.2 1644.78
  5063.0 1646.96  5076.1 1647.64  5118.1 1652.46  5159.4 1654.25  5266.2 1655.98
  5611.7 1655.81  5657.0 1657.42  5706.2 1663.97  5755.9 1666.22  5787.7 1667.79
#Mann=7,-1,0
  4626.1    0.07       0  4930.4   0.035       0  4938.2    0.07       0
  5011.9    0.07       0  5049.7    0.07       0  5051.2   0.035       0
  5755.9    0.07       0
Bank Sta=5011.9,5049.7
Exp/Cntr=0.3,0.1

Type RM Length L Ch R = 1,35990,120,120,120
BEGIN DESCRIPTION:
Mapping XS 79581d95
END DESCRIPTION:
XS GIS Cut Line= 3
      1643853.11      6952127.10      1644054.89      6952200.00
      1644721.21      6952402.62
#Sta/Elev= 30
  4783.9 1677.53  4807.2 1676.69  4826.9 1674.59  4832.2 1673.80  4849.7 1668.70
  4857.6 1667.44  4902.9 1662.67  4918.9 1659.51  4949.6 1655.99  4974.9 1646.54
  4995.9 1642.29  5001.1 1642.29  5006.3 1640.32  5025.5 1639.41  5026.5 1638.91
  5062.3 1638.91  5063.3 1639.41  5071.7 1639.62  5077.2 1642.26  5082.5 1641.93
  5110.1 1648.48  5129.3 1650.37  5143.0 1651.67  5267.7 1654.27  5287.3 1654.34
  5421.6 1654.13  5563.5 1654.86  5583.9 1654.25  5678.5 1656.47  5694.9 1656.82
#Mann=7,-1,0
  4783.9    0.07       0  5025.5    0.07       0  5063.3    0.07       0
  5129.3   0.035       0  5267.7    0.07       0  5287.3   0.035       0
  5678.5    0.07       0
Bank Sta=5025.5,5063.3
Exp/Cntr=0.3,0.1

Type RM Length L Ch R = 1,35870,537,537,537
BEGIN DESCRIPTION:
Mapping XS 3e84752f
END DESCRIPTION:
XS GIS Cut Line= 3
      1643800.98      6952265.10      1644005.41      6952304.16
      1644690.11      6952526.76
#Sta/Elev= 30
  4792.2 1677.48  4838.2 1676.08  4847.2 1675.23  4874.5 1668.60  4885.2 1666.49
  4942.4 1660.07  4949.0 1658.38  4969.4 1654.84  4989.4 1648.38  4991.5 1643.88
  4992.5 1643.38  5028.3 1643.38  5029.3 1643.88  5032.8 1646.98  5052.5 1646.58
  5059.5 1646.96  5084.0 1645.98  5091.4 1647.00  5096.7 1646.35  5115.6 1648.55
  5123.4 1648.32  5147.1 1650.85  5192.5 1651.44  5210.2 1652.31  5273.3 1653.84
  5536.2 1653.99  5645.0 1654.78  5681.6 1655.54  5714.9 1656.23  5720.3 1656.87
#Mann=5,-1,0
  4792.2    0.07       0  4874.5   0.035       0  4991.5   0.035       0
  5029.3   0.035       0  5681.6    0.07       0
Bank Sta=4991.5,5029.3
Exp/Cntr=0.3,0.1

Type RM Length L Ch R = 1,35333,439,439,439
BEGIN DESCRIPTION:
Mapping XS a5bc224d
END DESCRIPTION:
XS GIS Cut Line= 3
      1643597.60      6952729.30      1643903.59      6952781.38
      1644651.10      6952928.28
#Sta/Elev= 30
  4690.3 1680.32  4720.2 1678.43  4828.1 1674.76  4860.1 1670.45  4888.3 1665.07
  4893.4 1664.90  4901.9 1662.97  4921.0 1660.07  4953.6 1652.62  4961.5 1648.70
  4971.7 1644.61  4973.1 1642.07  4974.0 1641.57  5009.9 1641.57  5010.9 1642.07
  5013.3 1643.20  5022.5 1644.31  5064.7 1644.35  5093.8 1647.89  5111.0 1649.23
  5144.8 1649.41  5162.4 1650.47  5256.9 1651.94  5348.6 1652.56  5493.4 1652.61
  5603.4 1652.91  5705.3 1654.67  5725.7 1656.18  5746.1 1659.62  5762.5 1663.64
#Mann=6,-1,0
  4690.3   0.035       0  4720.2    0.07       0  4901.9   0.035       0
  4973.1   0.035       0  5010.9   0.035       0  5493.4    0.07       0
Bank Sta=4973.1,5010.9
Exp/Cntr=0.3,0.1

Type RM Length L Ch R = 1,34894,112,112,112
BEGIN DESCRIPTION:
Mapping XS 9f7ad3ed
END DESCRIPTION:
XS GIS Cut Line= 3
      1643618.27      6953082.46      1643855.92      6953205.08
      1644594.62      6953455.45
#Sta/Elev= 30
  4733.1 1669.80  4763.2 1664.68  4811.3 1659.14  4830.7 1657.98  4839.8 1656.82
  4853.2 1654.61  4867.6 1650.97  4906.3 1646.27  4928.5 1642.46  4931.6 1636.76
  4932.6 1636.26  4968.6 1636.26  4969.6 1636.76  4978.4 1638.30  4988.2 1638.43
  4998.3 1640.87  5002.7 1640.87  5010.1 1642.65  5020.3 1646.41  5031.2 1647.97
  5088.4 1649.24  5114.5 1648.95  5168.5 1649.93  5591.0 1653.33  5646.9 1654.87
  5674.7 1656.34  5717.5 1661.28  5764.6 1663.67  5777.5 1664.71  5780.5 1664.79
#Mann=7,-1,0
  4733.1    0.07       0  4811.3   0.035       0  4931.6   0.035       0
  4969.6   0.035       0  5646.9    0.07       0  5764.6   0.035       0
  5777.5    0.07       0
Bank Sta=4931.6,4969.6
Exp/Cntr=0.3,0.1

Type RM Length L Ch R = 1,34782,321,321,321
BEGIN DESCRIPTION:
Mapping XS f90b5864
END DESCRIPTION:
XS GIS Cut Line= 4
      1643549.96      6953233.30      1643755.01      6953284.29
      1643798.41      6953295.14      1644570.62      6953530.80
#Sta/Elev= 30
  4744.6 1667.69  4749.8 1666.19  4785.3 1661.29  4801.3 1657.93  4821.5 1656.63
  4839.0 1654.01  4868.0 1649.11  4904.2 1647.51  4914.7 1645.50  4945.5 1643.94
  4950.6 1644.50  4953.3 1642.14  4957.5 1641.70  4958.5 1641.20  4994.5 1641.20
  4995.5 1641.70  4996.3 1644.02  5025.4 1641.89  5049.3 1646.39  5063.4 1648.23
  5232.7 1649.97  5603.5 1652.01  5658.8 1653.33  5680.2 1654.32  5697.6 1657.30
  5713.0 1658.92  5718.5 1660.82  5739.4 1661.28  5800.4 1664.50  5808.0 1665.29
#Mann=6,-1,0
  4744.6    0.07       0  4839.0   0.035       0  4957.5   0.035       0
  4995.5   0.035       0  5658.8    0.07       0  5800.4   0.035       0
Bank Sta=4957.5,4995.5
Exp/Cntr=0.3,0.1

Type RM Length L Ch R = 1,34461,282,282,282
BEGIN DESCRIPTION:
Mapping XS b0e1b639
END DESCRIPTION:
XS GIS Cut Line= 3
      1643347.24      6953465.06      1643703.10      6953584.40
      1644471.14      6953850.91
#Sta/Elev= 30
  4626.0 1675.58  4634.2 1674.75  4676.4 1673.70  4697.5 1671.45  4708.0 1669.60
  4713.6 1667.38  4739.7 1662.17  4745.1 1660.47  4771.3 1656.80  4776.7 1654.95
  4802.9 1651.56  4807.9 1649.23  4855.7 1646.56  4902.9 1645.28  4919.0 1645.47
  4929.1 1644.62  4960.7 1645.68  4971.7 1644.36  4978.5 1640.75  4979.5 1640.25
  5015.5 1640.25  5016.5 1640.75  5023.4 1642.94  5035.1 1645.12  5054.5 1647.74
  5272.4 1647.71  5510.9 1650.31  5617.3 1652.32  5723.1 1655.28  5814.3 1661.42
#Mann=4,-1,0
  4626.0    0.07       0  4807.9   0.035       0  4978.5   0.035       0
  5016.5   0.035       0
Bank Sta=4978.5,5016.5
Exp/Cntr=0.3,0.1

Type RM Length L Ch R = 1,34179,412,412,412
BEGIN DESCRIPTION:
Mapping XS c8b9ec8d
END DESCRIPTION:
XS GIS Cut Line= 3
      1643230.00      6953563.00      1643538.58      6953805.08
      1644015.73      6954157.35
#Sta/Elev= 30
  4607.8 1675.72  4622.3 1675.56  4643.1 1674.35  4678.3 1674.01  4686.4 1674.48
  4692.8 1673.62  4721.7 1672.98  4736.2 1671.66  4757.0 1668.15  4785.9 1661.12
  4806.7 1658.07  4814.2 1655.36  4835.6 1652.44  4850.1 1648.84  4856.4 1648.05
  4906.5 1645.30  4914.2 1645.78  4949.5 1642.69  4964.0 1644.59  4978.4 1643.96
  5001.4 1641.76  5002.4 1641.26  5038.5 1641.26  5039.5 1641.76  5043.0 1643.72
  5078.5 1645.64  5114.0 1645.47  5157.1 1646.93  5235.1 1646.71  5593.1 1653.30
#Mann=4,-1,0
  4607.8    0.07       0  4814.2   0.035       0  5001.4   0.035       0
  5039.5   0.035       0
Bank Sta=5001.4,5039.5
Exp/Cntr=0.3,0.1

Type RM Length L Ch R = 1,33767,395,395,395
BEGIN DESCRIPTION:
Mapping XS a6f260d3
END DESCRIPTION:
XS GIS Cut Line= 3
      1642939.34      6953737.20      1643213.53      6954034.70
      1643980.55      6954185.06
#Sta/Elev= 30
  4597.9 1661.54  4613.2 1662.15  4673.2 1662.15  4699.1 1660.88  4722.5 1660.81
  4772.5 1657.22  4779.3 1657.64  4843.3 1654.17  4857.4 1654.52  4864.3 1653.30
  4885.3 1652.75  4935.5 1647.35  4942.0 1647.01  4956.2 1643.75  4958.7 1639.97
  4959.7 1639.47  4996.8 1639.97  4998.7 1641.53  5001.3 1641.73  5042.6 1641.63
  5099.2 1644.22  5126.3 1643.42  5218.0 1646.50  5268.9 1646.99  5361.6 1645.57
  5421.8 1642.65  5442.2 1643.94  5459.5 1646.53  5493.1 1647.54  5784.1 1653.16
#Mann=6,-1,0
  4597.9    0.07       0  4613.2    0.16       0  4699.1    0.07       0
  4935.5   0.035       0  4958.7   0.035       0  4996.8   0.035       0
Bank Sta=4958.7,4996.8
Exp/Cntr=0.3,0.1

Type RM Length L Ch R = 1,33372,401,401,401
BEGIN DESCRIPTION:
Mapping XS f6cba980
END DESCRIPTION:
XS GIS Cut Line= 4
      1642703.90      6953838.81      1643048.29      6954155.66
      1643355.37      6954367.80      1643756.42      6954745.93
#Sta/Elev= 30
  4158.8 1644.96  4314.6 1646.45  4343.0 1645.82  4505.7 1645.50  4661.3 1646.03
  4683.5 1645.17  4691.0 1645.77  4705.9 1645.27  4756.5 1645.79  4855.3 1644.17
  4870.2 1643.52  4899.9 1640.17  4906.0 1640.61  4926.9 1639.52  4963.1 1640.32
  4971.6 1640.03  4973.1 1638.48  4974.1 1637.98  5011.9 1638.48  5021.1 1639.70
  5035.3 1644.25  5063.6 1646.08  5077.8 1645.73  5098.8 1647.38  5282.9 1650.99
  5424.5 1654.80  5452.8 1654.55  5473.9 1656.03  5497.8 1656.22  5551.2 1657.34
#Mann=4,-1,0
  4158.8   0.035       0  4973.1   0.035       0  5011.9   0.035       0
  5497.8    0.07       0
Bank Sta=4973.1,5011.9
Exp/Cntr=0.3,0.1

Type RM Length L Ch R = 1,32971,276,276,276
BEGIN DESCRIPTION:
Mapping XS ee1768a1
END DESCRIPTION:
XS GIS Cut Line= 4
      1642716.94      6953971.21      1642970.84      6954266.34
      1643099.17      6954646.44      1643142.13      6954904.19
#Sta/Elev= 30
  4209.5 1644.75  4340.3 1645.66  4581.7 1644.59  4706.1 1645.16  4716.3 1644.06
  4721.6 1644.85  4747.8 1644.77  4753.1 1643.63  4769.4 1643.55  4784.5 1644.33
  4801.1 1643.57  4853.9 1643.31  4878.9 1643.92  4910.4 1643.58  4948.9 1641.93
  4973.3 1642.16  4978.8 1637.75  4979.8 1637.25  5017.6 1637.75  5021.9 1638.63
  5032.0 1638.97  5072.5 1646.12  5103.0 1650.07  5143.5 1650.39  5163.8 1652.77
  5188.3 1654.08  5214.5 1657.63  5244.1 1659.94  5249.2 1659.73  5261.3 1661.65
#Mann=3,-1,0
  4209.5   0.035       0  4978.8   0.035       0  5017.6   0.035       0
Bank Sta=4978.8,5017.6
Exp/Cntr=0.3,0.1

Type RM Length L Ch R = 1,32695,340,340,340
BEGIN DESCRIPTION:
Mapping XS 843f90ff
END DESCRIPTION:
XS GIS Cut Line= 4
      1642706.10      6954003.79      1642859.65      6954229.26
      1642852.63      6954642.01      1642838.93      6954828.41
#Sta/Elev= 30
  4314.4 1644.87  4338.4 1644.69  4367.9 1645.11  4431.2 1645.23  4482.0 1644.93
  4503.0 1645.33  4511.9 1644.88  4645.9 1643.79  4756.0 1644.46  4816.0 1643.88
  4836.0 1643.17  4866.0 1642.94  4906.0 1641.86  4926.0 1642.37  4946.0 1642.18
  4966.0 1639.41  4966.6 1636.10  4967.6 1635.60  5004.4 1635.60  5005.4 1636.10
  5006.0 1638.14  5016.0 1638.77  5038.5 1637.73  5046.1 1638.93  5056.1 1640.87
  5076.2 1647.61  5096.2 1651.97  5106.3 1653.59  5126.3 1655.82  5186.9 1659.35
#Mann=3,-1,0
  4314.4   0.035       0  4966.6    0.07       0  5005.4    0.07       0
Bank Sta=4966.6,5005.4
Exp/Cntr=0.3,0.1

Type RM Length L Ch R = 1,32355,316,316,316
BEGIN DESCRIPTION:
Mapping XS 700c4e09
END DESCRIPTION:
XS GIS Cut Line= 3
      1642772.71      6954126.13      1642561.58      6954501.63
      1642492.56      6954668.32
#Sta/Elev= 30
  4573.0 1645.19  4735.8 1643.49  4793.1 1642.32  4800.9 1641.78  4822.6 1642.06
  4844.3 1641.40  4865.9 1642.47  4887.6 1642.51  4903.6 1643.52  4909.3 1642.54
  4931.0 1641.97  4946.9 1639.79  4961.1 1636.15  4976.7 1633.79  4990.2 1632.68
  4992.6 1630.31  4993.6 1629.81  5030.4 1629.81  5031.4 1630.31  5035.9 1634.47
  5043.2 1636.73  5054.0 1639.16  5059.8 1639.67  5065.2 1641.35  5097.3 1648.61
  5129.7 1652.60  5151.4 1655.89  5166.2 1656.77  5173.0 1658.20  5184.2 1659.18
#Mann=4,-1,0
  4573.0   0.035       0  4961.1    0.07       0  4992.6    0.07       0
  5031.4    0.07       0
Bank Sta=4992.6,5031.4
Exp/Cntr=0.3,0.1

Type RM Length L Ch R = 1,32039,319,319,319
BEGIN DESCRIPTION:
Mapping XS 142a36ee
END DESCRIPTION:
XS GIS Cut Line= 3
      1642543.52      6953976.85      1642284.24      6954372.72
      1642186.01      6954534.28
#Sta/Elev= 30
  4530.6 1643.99  4675.4 1643.83  4682.2 1642.42  4688.2 1642.56  4718.4 1639.64
  4739.5 1638.64  4775.7 1640.01  4811.8 1639.07  4863.1 1640.17  4869.1 1639.14
  4914.4 1639.45  4926.5 1635.34  4941.5 1632.14  4950.4 1631.19  4952.2 1629.94
  4953.2 1629.44  4991.1 1629.94  4998.6 1632.48  5003.8 1632.48  5013.9 1637.01
  5021.7 1639.02  5029.4 1642.11  5056.8 1648.69  5080.2 1650.62  5093.4 1653.16
  5115.3 1655.70  5130.2 1658.40  5151.5 1663.78  5155.5 1663.98  5192.9 1665.28
#Mann=4,-1,0
  4530.6   0.035       0  4952.2   0.035       0  4991.1   0.035       0
  5155.5    0.07       0
Bank Sta=4952.2,4991.1
Exp/Cntr=0.3,0.1

Type RM Length L Ch R = 1,31720,306,306,306
BEGIN DESCRIPTION:
Mapping XS c46e1f73
END DESCRIPTION:
XS GIS Cut Line= 3
      1642425.18      6953839.31      1642089.25      6954128.37
      1641931.68      6954336.72
#Sta/Elev= 30
  4560.7 1642.77  4638.3 1642.83  4666.5 1641.97  4703.6 1642.49  4822.6 1641.22
  4843.4 1639.79  4857.7 1636.05  4878.6 1634.45  4900.5 1634.32  4914.8 1636.07
  4929.0 1635.60  4949.9 1637.73  4964.1 1635.73  4978.4 1635.27  4983.9 1631.37
  4984.9 1630.87  5022.8 1631.37  5028.5 1633.16  5035.3 1633.35  5056.1 1639.95
  5070.7 1643.49  5091.5 1646.48  5106.0 1647.20  5149.7 1653.11  5166.9 1658.36
  5170.5 1659.72  5178.8 1660.65  5185.5 1662.59  5205.9 1664.63  5265.1 1666.41
#Mann=6,-1,0
  4560.7   0.035       0  4703.6    0.07       0  4983.9    0.07       0
  5022.8    0.07       0  5166.9   0.035       0  5185.5    0.07       0
Bank Sta=4983.9,5022.8
Exp/Cntr=0.3,0.1

Type RM Length L Ch R = 1,31414,396,396,396
BEGIN DESCRIPTION:
Mapping XS 854bcf12
END DESCRIPTION:
XS GIS Cut Line= 3
      1642313.95      6953697.82      1641901.64      6953893.12
      1641827.85      6954032.02
#Sta/Elev= 30
  4553.3 1642.14  4654.7 1641.29  4686.3 1640.97  4709.1 1641.61  4754.6 1641.22
  4845.5 1639.17  4868.3 1637.89  4891.0 1635.17  4919.3 1634.43  4959.3 1630.16
  4964.8 1628.94  4972.6 1628.37  4975.3 1627.08  4976.3 1626.58  5013.2 1626.58
  5014.2 1627.08  5016.9 1631.20  5033.2 1632.98  5038.8 1634.99  5055.2 1638.07
  5060.8 1640.13  5071.5 1641.51  5077.1 1643.53  5093.5 1646.27  5099.1 1648.04
  5121.1 1651.27  5150.9 1653.36  5159.4 1656.83  5164.5 1658.20  5166.8 1658.20
#Mann=4,-1,0
  4553.3   0.035       0  4654.7    0.07       0  4975.3    0.07       0
  5014.2    0.07       0
Bank Sta=4975.3,5014.2
Exp/Cntr=0.3,0.1

Type RM Length L Ch R = 1,31018,403,403,403
BEGIN DESCRIPTION:
Mapping XS 2f514460
END DESCRIPTION:
XS GIS Cut Line= 3
      1642316.15      6953435.22      1641751.90      6953548.07
      1641429.28      6953600.04
#Sta/Elev= 30
  4427.3 1641.33  4510.1 1641.02  4612.0 1639.50  4618.5 1640.06  4623.6 1639.60
  4632.4 1640.85  4642.6 1640.84  4663.0 1639.62  4725.6 1640.12  4858.7 1638.06
  4907.8 1636.98  4929.6 1635.66  4948.6 1632.90  4979.1 1625.19  4980.1 1624.69
  5017.0 1624.69  5018.0 1625.19  5019.8 1627.50  5029.3 1632.58  5034.4 1632.92
  5040.1 1636.67  5050.2 1638.26  5070.5 1643.79  5101.3 1648.79  5121.1 1654.92
  5131.3 1656.82  5171.8 1658.68  5212.3 1658.82  5242.7 1660.54  5329.5 1662.02
#Mann=4,-1,0
  4427.3   0.035       0  4858.7    0.07       0  4979.1    0.07       0
  5018.0    0.07       0
Bank Sta=4979.1,5018
Exp/Cntr=0.3,0.1

Type RM Length L Ch R = 1,30615,493,493,493
BEGIN DESCRIPTION:
Mapping XS 19621ffe
END DESCRIPTION:
XS GIS Cut Line= 3
      1642203.45      6953033.58      1641649.65      6953177.67
      1641420.52      6953271.41
#Sta/Elev= 30
  4433.1 1640.56  4483.2 1639.49  4555.5 1639.74  4617.5 1638.46  4671.7 1638.76
  4712.2 1637.29  4747.6 1638.89  4752.7 1638.07  4793.3 1638.31  4864.0 1637.18
  4869.1 1637.21  4886.1 1641.00  4909.7 1639.29  4927.5 1634.62  4945.0 1631.30
  4950.2 1631.04  4958.5 1628.78  4980.3 1625.00  4981.3 1624.50  5019.3 1625.00
  5032.0 1625.85  5047.0 1629.61  5053.6 1633.05  5071.0 1638.25  5086.0 1640.81
  5107.6 1645.92  5118.4 1647.79  5148.3 1650.25  5183.3 1652.68  5252.9 1654.03
#Mann=4,-1,0
  4433.1   0.035       0  4980.3   0.035       0  5019.3   0.035       0
  5148.3    0.07       0
Bank Sta=4980.3,5019.3
Exp/Cntr=0.3,0.1

Type RM Length L Ch R = 1,30122,147,147,147
BEGIN DESCRIPTION:
Mapping XS c99fae47
END DESCRIPTION:
XS GIS Cut Line= 4
      1642366.83      6952300.65      1641630.55      6952654.67
      1641449.99      6952753.63      1640845.82      6953000.16
#Sta/Elev= 30
  3981.4 1666.53  4010.5 1664.35  4027.6 1661.48  4038.9 1657.99  4061.3 1655.44
  4123.7 1651.40  4205.3 1640.77  4252.9 1639.15  4632.8 1636.22  4818.8 1636.22
  4878.5 1634.02  4930.1 1627.93  4938.2 1627.71  4943.9 1626.05  4968.0 1625.10
  4969.0 1624.60  5007.0 1625.10  5027.5 1625.80  5051.5 1629.30  5086.3 1636.77
  5105.0 1637.63  5110.4 1639.37  5117.7 1638.06  5128.5 1637.76  5193.3 1639.73
  5366.1 1642.43  5401.8 1644.82  5508.7 1647.22  5592.9 1647.80  5656.8 1647.05
#Mann=4,-1,0
  3981.4    0.07       0  4252.9   0.035       0  4968.0   0.035       0
  5007.0   0.035       0
Bank Sta=4968,5007
Exp/Cntr=0.3,0.1

Type RM Length L Ch R = 1,29975,168,168,168
BEGIN DESCRIPTION:
Mapping XS 535df2b4
END DESCRIPTION:
XS GIS Cut Line= 3
      1642297.37      6952210.38      1641387.49      6952625.15
      1640849.62      6952809.07
#Sta/Elev= 30
  4002.9 1666.52  4049.5 1664.77  4084.7 1657.12  4148.4 1651.97  4246.0 1639.31
  4272.6 1638.34  4691.9 1635.55  4692.9 1635.05  4730.9 1635.55  4734.4 1637.80
  4751.9 1640.67  4780.5 1640.25  4786.0 1644.06  4803.5 1641.27  4809.0 1645.62
  4826.6 1642.25  4832.1 1646.19  4849.6 1642.72  4855.1 1646.41  4859.9 1645.69
  4872.7 1644.14  4878.2 1647.91  4901.2 1647.28  4952.8 1650.14  5050.3 1649.51
  5068.9 1647.17  5100.6 1637.83  5118.1 1636.59  5425.9 1641.08  5571.3 1640.72
#Mann=6,-1,0
  4002.9    0.07       0  4272.6   0.035       0  4691.9    0.07       0
  4730.9   0.035       0  4859.9    0.07       0  5050.3   0.035       0
Bank Sta=4691.9,4730.9
Exp/Cntr=0.3,0.1

Type RM Length L Ch R = 1,29807,759,759,759
BEGIN DESCRIPTION:
Mapping XS d933e94d
END DESCRIPTION:
XS GIS Cut Line= 5
      1642200.18      6952151.34      1641569.78      6952451.54
      1641340.62      6952472.38      1641243.40      6952474.11
      1640807.63      6952673.77
#Sta/Elev= 30
  4070.0 1664.30  4086.8 1662.37  4117.4 1656.49  4140.1 1653.35  4213.8 1646.44
  4219.7 1645.08  4230.8 1644.59  4264.7 1639.76  4294.3 1638.73  4372.7 1636.89
  4491.8 1635.68  4684.9 1635.49  4718.1 1635.90  4740.3 1641.53  4747.1 1641.66
  4752.6 1641.33  4768.1 1635.84  4953.8 1631.48  4973.9 1628.40  4974.1 1624.94
  4975.1 1624.44  5013.1 1624.94  5014.0 1626.41  5036.1 1627.25  5043.0 1628.45
  5064.0 1633.46  5097.8 1634.73  5193.6 1634.81  5383.1 1637.90  5574.9 1638.91
#Mann=6,-1,0
  4070.0    0.07       0  4294.3   0.035       0  4974.1   0.035       0
  5013.1   0.035       0  5043.0    0.07       0  5097.8   0.035       0
Bank Sta=4974.1,5013.1
Exp/Cntr=0.3,0.1

Type RM Length L Ch R = 1,29048,464,464,464
BEGIN DESCRIPTION:
Mapping XS ae934f3d
END DESCRIPTION:
XS GIS Cut Line= 3
      1641126.09      6951594.57      1641008.91      6951890.13
      1640858.34      6952524.87
#Sta/Elev= 30
  4685.2 1662.30  4742.7 1660.69  4764.2 1658.72  4787.1 1658.98  4806.0 1656.56
  4811.4 1656.89  4818.0 1655.53  4850.2 1654.74  4860.1 1652.53  4865.5 1652.87
  4871.8 1649.73  4889.8 1644.17  4895.2 1644.45  4904.0 1642.07  4919.5 1640.47
  4936.3 1636.29  4943.8 1633.17  4949.2 1633.11  4957.8 1630.10  4973.5 1621.92
  4997.3 1623.21  5001.7 1622.93  5001.9 1618.89  5002.9 1618.39  5041.1 1618.89
  5044.5 1621.07  5072.9 1631.00  5086.7 1631.90  5350.4 1632.83  5655.5 1637.30
#Mann=4,-1,0
  4685.2    0.07       0  4997.3   0.035       0  5001.9   0.035       0
  5041.1   0.035       0
Bank Sta=5001.9,5041.1
Exp/Cntr=0.3,0.1

Type RM Length L Ch R = 1,28584,290,290,290
BEGIN DESCRIPTION:
Mapping XS 8789b622
END DESCRIPTION:
XS GIS Cut Line= 3
      1640491.98      6951640.12      1640563.60      6951943.51
      1640709.43      6952560.68
#Sta/Elev= 30
  4694.0 1652.34  4743.2 1650.33  4755.3 1650.78  4804.8 1649.68  4860.4 1646.00
  4866.5 1643.27  4876.8 1641.11  4887.0 1637.49  4902.7 1634.08  4907.9 1633.84
  4938.4 1627.57  4945.0 1625.64  4969.2 1622.21  4979.5 1618.74  4980.5 1617.57
  4981.5 1617.07  5018.7 1617.07  5019.7 1617.57  5034.8 1619.44  5061.7 1628.09
  5102.8 1629.74  5195.3 1630.00  5204.0 1630.56  5209.1 1629.86  5246.3 1631.24
  5420.6 1634.12  5431.6 1634.82  5534.4 1636.14  5552.6 1635.80  5639.9 1637.58
#Mann=4,-1,0
  4694.0   0.035       0  4755.3    0.07       0  4980.5   0.035       0
  5019.7   0.035       0
Bank Sta=4980.5,5019.7
Exp/Cntr=0.3,0.1

Type RM Length L Ch R = 1,28294,283,283,283
BEGIN DESCRIPTION:
Mapping XS 767cc703
END DESCRIPTION:
XS GIS Cut Line= 3
      1640157.58      6951751.66      1640304.05      6952035.92
      1640518.56      6952553.77
#Sta/Elev= 30
  4682.1 1649.43  4765.7 1648.77  4790.5 1647.96  4818.5 1648.33  4824.2 1647.51
  4840.7 1647.12  4879.4 1644.21  4891.7 1639.80  4914.2 1629.99  4929.3 1627.70
  4951.5 1620.40  4954.0 1615.51  4955.0 1615.01  4992.2 1615.01  4993.2 1615.51
  5000.2 1620.43  5018.9 1621.08  5025.8 1619.28  5036.6 1620.97  5042.8 1624.38
  5045.8 1624.77  5058.2 1626.87  5066.7 1627.60  5119.9 1628.23  5134.0 1629.41
  5188.1 1630.37  5226.2 1630.22  5296.4 1631.13  5361.9 1632.83  5562.4 1635.98
#Mann=5,-1,0
  4682.1   0.035       0  4765.7    0.07       0  4954.0    0.07       0
  4993.2    0.07       0  5045.8   0.035       0
Bank Sta=4954,4993.2
Exp/Cntr=0.3,0.1

Type RM Length L Ch R = 1,28011,324,324,324
BEGIN DESCRIPTION:
Mapping XS 35a03b1a
END DESCRIPTION:
XS GIS Cut Line= 3
      1639877.92      6951855.10      1640054.99      6952138.06
      1640329.28      6952632.82
#Sta/Elev= 30
  4670.5 1645.88  4692.4 1645.68  4713.7 1646.34  4753.0 1645.93  4780.1 1645.76
  4786.8 1645.11  4844.5 1643.91  4865.7 1642.94  4874.5 1641.90  4881.1 1639.53
  4887.0 1638.61  4896.4 1635.28  4902.3 1634.40  4909.9 1631.70  4938.8 1625.85
  4945.2 1622.56  4949.2 1616.32  4950.2 1615.82  4987.4 1615.82  4988.4 1616.32
  5012.3 1616.74  5027.1 1618.15  5034.0 1621.51  5039.8 1623.05  5050.0 1625.41
  5061.5 1626.59  5196.6 1629.21  5327.0 1630.29  5554.8 1635.16  5570.0 1634.92
#Mann=4,-1,0
  4670.5   0.035       0  4753.0    0.07       0  4949.2   0.035       0
  4988.4   0.035       0
Bank Sta=4949.2,4988.4
Exp/Cntr=0.3,0.1

Type RM Length L Ch R = 1,27687,287,287,287
BEGIN DESCRIPTION:
Mapping XS 7cf0c543
END DESCRIPTION:
XS GIS Cut Line= 3
      1639571.03      6951961.38      1639761.15      6952232.24
      1640093.17      6952672.32
#Sta/Elev= 30
  4669.5 1640.87  4671.7 1640.86  4720.1 1641.38  4741.1 1640.64  4755.9 1641.49
  4799.8 1640.49  4836.0 1638.20  4842.1 1638.49  4848.6 1637.36  4863.1 1636.91
  4877.9 1635.43  4892.7 1632.01  4907.5 1630.60  4921.9 1628.07  4928.4 1626.34
  4949.3 1623.97  4958.0 1621.36  4959.4 1616.12  4960.4 1615.62  4998.6 1616.12
  5049.9 1617.59  5057.7 1618.79  5064.5 1622.28  5070.7 1623.72  5085.3 1625.64
  5129.0 1625.65  5220.6 1627.48  5328.8 1627.20  5478.7 1631.40  5551.7 1632.68
#Mann=5,-1,0
  4669.5   0.035       0  4671.7    0.07       0  4921.9   0.035       0
  4959.4   0.035       0  4998.6   0.035       0
Bank Sta=4959.4,4998.6
Exp/Cntr=0.3,0.1

Type RM Length L Ch R = 1,27400,334,334,334
BEGIN DESCRIPTION:
Mapping XS bf7695ee
END DESCRIPTION:
XS GIS Cut Line= 3
      1639403.10      6952056.50      1639521.57      6952372.87
      1639842.27      6952884.43
#Sta/Elev= 30
  4663.9 1633.67  4687.9 1634.66  4743.1 1633.22  4783.0 1629.64  4798.3 1629.15
  4823.2 1626.01  4836.4 1627.20  4868.8 1625.51  4889.7 1624.12  4939.0 1622.76
  4944.3 1621.08  4953.8 1619.29  4963.9 1618.77  4985.9 1618.97  4999.5 1620.80
  5066.8 1619.53  5079.3 1621.05  5102.2 1619.30  5105.6 1617.07  5106.6 1616.57
  5143.8 1616.57  5144.8 1617.07  5146.4 1624.19  5161.2 1625.63  5232.0 1626.23
  5240.7 1626.78  5377.4 1627.16  5398.6 1628.10  5479.9 1628.89  5605.5 1632.83
#Mann=4,-1,0
  4663.9    0.07       0  4868.8   0.035       0  5105.6   0.035       0
  5144.8   0.035       0
Bank Sta=5105.6,5144.8
Exp/Cntr=0.3,0.1

Type RM Length L Ch R = 1,27066,243,243,243
BEGIN DESCRIPTION:
Mapping XS 7a659148
END DESCRIPTION:
XS GIS Cut Line= 3
      1639290.12      6952254.47      1639350.98      6952639.49
      1639474.44      6953024.79
#Sta/Elev= 30
  4614.2 1625.93  4648.1 1625.50  4708.9 1622.85  4769.6 1622.01  4789.9 1621.26
  4850.6 1621.77  4872.8 1622.23  4881.0 1622.86  4911.4 1622.34  4930.1 1620.92
  4951.9 1617.74  4962.0 1616.96  4962.5 1615.83  4963.5 1615.33  5000.9 1615.33
  5001.9 1615.83  5004.0 1616.44  5012.9 1616.20  5023.4 1618.49  5068.5 1620.35
  5092.7 1622.35  5100.6 1622.59  5107.4 1624.26  5127.5 1625.77  5132.8 1625.59
  5159.7 1627.29  5197.1 1628.90  5363.0 1633.56  5395.1 1634.88  5408.6 1636.47
#Mann=4,-1,0
  4614.2   0.035       0  4962.5    0.07       0  5001.9   0.035       0
  5092.7   0.035       0
Bank Sta=4962.5,5001.9
Exp/Cntr=0.3,0.1

Type RM Length L Ch R = 1,26823,189,189,189
BEGIN DESCRIPTION:
Mapping XS 4eea124f
END DESCRIPTION:
XS GIS Cut Line= 3
      1639226.32      6952289.64      1639106.84      6952638.40
      1639033.61      6952952.42
#Sta/Elev= 30
  4635.2 1625.44  4688.6 1624.49  4707.5 1623.61  4714.6 1622.59  4728.6 1622.21
  4745.9 1622.47  4770.9 1621.94  4808.4 1622.64  4834.3 1621.79  4839.7 1621.09
  4902.3 1620.90  4928.3 1619.48  4933.6 1618.52  4940.0 1614.54  4950.6 1613.58
  4971.1 1613.38  4972.1 1612.88  5009.5 1612.88  5010.5 1613.38  5013.7 1619.98
  5024.0 1623.24  5036.7 1624.39  5085.6 1624.05  5126.9 1624.66  5169.5 1626.38
  5206.9 1628.57  5291.0 1631.10  5297.1 1631.84  5302.3 1631.25  5326.3 1631.83
#Mann=3,-1,0
  4635.2   0.035       0  4971.1   0.035       0  5010.5   0.035       0
Bank Sta=4971.1,5010.5
Exp/Cntr=0.3,0.1

Type RM Length L Ch R = 1,26634,27,27,27
BEGIN DESCRIPTION:
Mapping XS 3de640db
END DESCRIPTION:
XS GIS Cut Line= 4
      1639088.13      6952337.13      1638938.74      6952571.93
      1638920.21      6952592.83      1638937.49      6952854.23
#Sta/Elev= 30
  4721.7 1625.00  4738.7 1624.96  4753.9 1623.87  4759.8 1624.22  4769.2 1623.32
  4790.3 1622.43  4811.5 1622.16  4826.7 1621.06  4947.9 1620.44  4957.1 1618.93
  4963.1 1618.90  4971.6 1616.15  4973.8 1613.00  4974.8 1612.50  5012.2 1612.50
  5013.2 1613.00  5014.0 1614.00  5027.9 1613.55  5043.1 1614.47  5063.2 1621.03
  5073.2 1622.79  5083.2 1623.55  5103.3 1623.83  5143.4 1622.97  5153.4 1622.33
  5177.4 1622.76  5213.5 1625.20  5233.5 1627.09  5263.6 1627.87  5289.9 1629.18
#Mann=3,-1,0
  4721.7   0.035       0  4973.8   0.035       0  5013.2   0.035       0
Bank Sta=4973.8,5013.2
Exp/Cntr=0.3,0.1

Type RM Length L Ch R = 1,26607,24,24,24
BEGIN DESCRIPTION:
Mapping XS 7def3620
END DESCRIPTION:
XS GIS Cut Line= 4
      1639049.12      6952312.09      1638919.70      6952553.14
      1638899.60      6952577.64      1638892.00      6952853.15
#Sta/Elev= 30
  4726.4 1625.70  4791.7 1624.35  4808.0 1623.41  4835.6 1622.78  4846.2 1622.10
  4851.8 1622.53  4858.0 1621.46  4880.7 1620.35  4917.6 1620.03  4933.8 1620.47
  4948.8 1620.34  4971.5 1618.62  4983.4 1616.87  5006.4 1618.36  5011.7 1616.38
  5012.7 1615.88  5050.1 1615.88  5051.1 1616.38  5052.1 1617.32  5072.1 1618.60
  5092.1 1622.68  5102.1 1623.51  5122.1 1623.60  5162.1 1621.82  5172.1 1621.99
  5202.1 1623.75  5222.1 1626.26  5242.1 1628.01  5302.2 1629.59  5307.3 1630.01
#Mann=3,-1,0
  4726.4   0.035       0  5011.7   0.035       0  5051.1   0.035       0
Bank Sta=5011.7,5051.1
Exp/Cntr=0.3,0.1

Type RM Length L Ch R = 1,26583,281,281,281
BEGIN DESCRIPTION:
Mapping XS a001fc05
END DESCRIPTION:
XS GIS Cut Line= 4
      1638995.93      6952317.55      1638901.77      6952538.58
      1638882.23      6952566.79      1638850.98      6952844.88
#Sta/Elev= 30
  4762.7 1625.27  4855.0 1623.09  4878.6 1621.23  4884.0 1621.45  4902.2 1620.07
  4931.3 1619.57  4960.3 1619.73  4978.5 1618.13  4984.0 1616.54  4999.9 1616.50
  5002.4 1615.85  5003.4 1615.35  5040.8 1615.35  5041.8 1615.85  5048.5 1616.65
  5055.4 1616.87  5068.7 1616.38  5088.8 1617.77  5098.9 1619.32  5108.9 1621.75
  5119.0 1623.30  5139.1 1623.66  5169.3 1621.63  5189.4 1621.89  5209.5 1623.31
  5219.6 1624.65  5235.5 1627.91  5240.5 1628.40  5259.9 1629.54  5317.1 1630.36
#Mann=3,-1,0
  4762.7   0.035       0  5002.4   0.035       0  5041.8   0.035       0
Bank Sta=5002.4,5041.8
Exp/Cntr=0.3,0.1

Type RM Length L Ch R = 1,26302,427,427,427
BEGIN DESCRIPTION:
Mapping XS 56fbaa73
END DESCRIPTION:
XS GIS Cut Line= 3
      1638638.74      6952014.30      1638655.02      6952447.25
      1638651.77      6952807.48
#Sta/Elev= 30
  4571.5 1634.07  4637.3 1631.66  4695.3 1626.15  4725.3 1624.49  4735.3 1624.65
  4765.3 1623.39  4775.3 1623.61  4828.4 1621.92  4865.4 1621.07  4870.8 1620.51
  4885.4 1620.67  4905.4 1618.89  4915.4 1615.64  4955.5 1616.05  4965.5 1615.53
  4975.5 1613.68  4995.5 1614.30  4999.9 1613.61  5015.7 1612.38  5016.7 1611.88
  5054.4 1611.88  5055.4 1612.38  5055.5 1613.67  5065.5 1615.86  5085.5 1621.37
  5097.6 1623.18  5156.1 1627.30  5205.5 1629.30  5255.1 1629.81  5365.0 1630.14
#Mann=9,-1,0
  4571.5    0.07       0  4637.3    0.16       0  4828.4   0.035       0
  4999.9    0.07       0  5015.7    0.07       0  5055.4    0.07       0
  5097.6   0.035       0  5156.1    0.07       0  5255.1   0.035       0
Bank Sta=5015.7,5055.4
Exp/Cntr=0.3,0.1

Type RM Length L Ch R = 1,25875,432,432,432
BEGIN DESCRIPTION:
Mapping XS 8e28cfe2
END DESCRIPTION:
XS GIS Cut Line= 3
      1638048.48      6952051.22      1638245.95      6952388.66
      1638430.73      6952839.27
#Sta/Elev= 30
  4610.3 1632.66  4681.9 1631.68  4757.4 1630.44  4773.1 1629.93  4788.8 1628.36
  4794.6 1628.61  4810.3 1627.18  4847.5 1626.60  4867.5 1620.55  4890.5 1615.39
  4906.2 1614.74  4927.6 1616.51  4942.6 1616.27  4949.1 1614.20  4954.9 1613.91
  4964.8 1611.05  4966.5 1607.78  4967.5 1607.28  5005.2 1607.28  5006.2 1607.78
  5009.0 1611.42  5038.3 1611.35  5054.6 1613.11  5062.3 1615.90  5067.7 1615.86
  5076.2 1618.86  5086.3 1619.73  5132.7 1620.63  5216.1 1621.52  5488.3 1626.75
#Mann=7,-1,0
  4610.3    0.16       0  4681.9    0.07       0  4867.5   0.035       0
  4966.5   0.035       0  5006.2   0.035       0  5132.7    0.07       0
  5216.1   0.035       0
Bank Sta=4966.5,5006.2
Exp/Cntr=0.3,0.1

Type RM Length L Ch R = 1,25443,331,331,331
BEGIN DESCRIPTION:
Mapping XS c2b1913b
END DESCRIPTION:
XS GIS Cut Line= 3
      1637642.76      6952450.40      1637909.69      6952636.59
      1638300.80      6952879.58
#Sta/Elev= 30
  4673.9 1630.34  4823.7 1628.29  4868.2 1626.84  4896.1 1625.00  4932.7 1623.52
  4939.7 1621.88  4945.8 1619.20  4954.5 1616.73  4960.6 1614.01  4969.2 1611.49
  4979.6 1610.39  4996.2 1609.64  4997.5 1608.95  4998.5 1608.45  5036.3 1608.45
  5037.3 1608.95  5040.9 1610.23  5054.0 1611.61  5063.5 1612.30  5076.2 1612.06
  5084.7 1612.55  5090.6 1613.23  5096.7 1614.81  5106.0 1617.68  5127.2 1618.18
  5142.6 1619.25  5153.9 1619.28  5215.8 1620.29  5279.5 1620.50  5459.8 1624.25
#Mann=6,-1,0
  4673.9    0.07       0  4979.6   0.035       0  4997.5   0.035       0
  5037.3   0.035       0  5096.7    0.07       0  5153.9   0.035       0
Bank Sta=4997.5,5037.3
Exp/Cntr=0.3,0.1

Type RM Length L Ch R = 1,25112,365,365,365
BEGIN DESCRIPTION:
Mapping XS 55eb3d9e
END DESCRIPTION:
XS GIS Cut Line= 3
      1637452.24      6952797.19      1637801.18      6952935.21
      1638208.50      6953103.08
#Sta/Elev= 30
  4624.4 1629.45  4631.1 1629.46  4744.6 1628.76  4833.8 1626.65  4874.7 1624.64
  4887.9 1623.17  4899.0 1619.20  4912.2 1615.33  4917.7 1613.03  4936.6 1608.80
  4960.7 1608.96  4962.3 1607.00  4963.3 1606.50  5001.1 1606.50  5002.1 1607.00
  5004.4 1607.78  5014.6 1607.96  5036.2 1611.35  5057.9 1612.95  5067.9 1612.58
  5090.3 1613.69  5097.3 1613.00  5111.9 1613.45  5121.2 1612.73  5133.6 1613.22
  5144.4 1614.76  5150.6 1617.15  5174.5 1618.90  5286.5 1620.48  5440.2 1624.14
#Mann=5,-1,0
  4624.4   0.035       0  4631.1    0.07       0  4899.0   0.035       0
  4962.3   0.035       0  5002.1   0.035       0
Bank Sta=4962.3,5002.1
Exp/Cntr=0.3,0.1

Type RM Length L Ch R = 1,24747,406,406,406
BEGIN DESCRIPTION:
Mapping XS c7efbef1
END DESCRIPTION:
XS GIS Cut Line= 3
      1637377.84      6953203.43      1637752.87      6953284.16
      1638209.94      6953389.64
#Sta/Elev= 30
  4617.2 1627.66  4655.2 1627.76  4666.6 1627.25  4798.4 1625.93  4804.4 1625.25
  4853.7 1623.64  4870.0 1622.28  4880.4 1619.99  4890.5 1617.40  4897.9 1613.99
  4903.0 1613.64  4910.9 1611.71  4931.4 1608.52  4952.4 1607.06  4962.1 1604.99
  4991.5 1605.54  4993.4 1604.21  4994.4 1603.71  5032.2 1603.71  5033.2 1604.21
  5033.8 1608.95  5039.5 1611.58  5054.3 1613.22  5082.3 1615.28  5136.4 1617.17
  5228.8 1618.85  5258.5 1621.66  5306.4 1623.46  5422.8 1624.36  5469.9 1625.07
#Mann=5,-1,0
  4617.2    0.07       0  4880.4   0.035       0  4993.4   0.035       0
  5033.2   0.035       0  5422.8    0.07       0
Bank Sta=4993.4,5033.2
Exp/Cntr=0.3,0.1

Type RM Length L Ch R = 1,24341,333,333,333
BEGIN DESCRIPTION:
Mapping XS 61ea7349
END DESCRIPTION:
XS GIS Cut Line= 3
      1637314.09      6953525.06      1637704.70      6953674.79
      1638130.89      6953829.41
#Sta/Elev= 30
  4582.2 1626.23  4711.2 1625.65  4832.4 1623.71  4848.4 1621.83  4850.7 1621.52
  4856.1 1621.86  4880.7 1613.29  4886.1 1612.87  4893.8 1611.16  4910.8 1609.38
  4925.9 1609.59  4940.8 1607.74  4947.3 1605.47  4958.0 1603.27  4970.8 1603.53
  4978.1 1602.01  4979.1 1601.51  5017.0 1601.51  5018.0 1602.01  5020.7 1604.58
  5026.0 1605.90  5032.8 1611.14  5043.4 1614.80  5051.3 1615.38  5117.9 1616.89
  5160.4 1616.94  5266.8 1618.86  5352.2 1619.86  5426.4 1623.08  5453.9 1625.30
#Mann=5,-1,0
  4582.2   0.035       0  4832.4    0.07       0  4848.4   0.035       0
  4978.1   0.035       0  5018.0   0.035       0
Bank Sta=4978.1,5018
Exp/Cntr=0.3,0.1

Type RM Length L Ch R = 1,24008,491,491,491
BEGIN DESCRIPTION:
Mapping XS e5532511
END DESCRIPTION:
XS GIS Cut Line= 3
      1637353.34      6953873.50      1637603.31      6953958.56
      1638108.51      6954102.65
#Sta/Elev= 30
  4734.5 1621.59  4783.7 1621.53  4826.1 1621.32  4852.1 1620.74  4857.4 1620.14
  4887.3 1619.93  4905.3 1620.26  4920.2 1619.37  4926.4 1617.30  4951.5 1611.70
  4968.6 1605.34  4977.6 1601.29  4995.4 1600.53  4996.4 1600.03  5034.3 1600.03
  5035.3 1600.53  5040.7 1602.80  5049.2 1606.48  5054.4 1607.25  5062.7 1609.96
  5073.1 1612.12  5104.3 1614.11  5145.9 1615.44  5235.3 1616.52  5379.6 1618.14
  5418.6 1619.57  5452.5 1621.50  5468.3 1624.40  5478.6 1625.53  5523.9 1627.84
#Mann=7,-1,0
  4734.5   0.035       0  4783.7    0.16       0  4887.3    0.07       0
  4995.4    0.07       0  5035.3    0.07       0  5040.7   0.035       0
  5235.3    0.07       0
Bank Sta=4995.4,5035.3
Exp/Cntr=0.3,0.1

Type RM Length L Ch R = 1,23517,427,427,427
BEGIN DESCRIPTION:
Mapping XS ebd70ad8
END DESCRIPTION:
XS GIS Cut Line= 3
      1637363.50      6954098.72      1637522.36      6954424.27
      1637705.43      6954603.44
#Sta/Elev= 30
  4639.9 1615.03  4647.0 1615.20  4722.8 1613.41  4750.9 1611.54  4835.5 1608.25
  4841.0 1607.26  4872.8 1606.53  4886.1 1607.04  4903.1 1605.55  4925.6 1605.21
  4948.1 1606.14  4972.6 1604.89  4976.2 1605.51  4993.2 1605.71  5001.4 1604.74
  5022.1 1603.93  5023.1 1603.43  5061.0 1603.43  5062.0 1603.93  5063.2 1608.02
  5084.8 1610.50  5091.4 1611.82  5126.9 1615.43  5133.9 1618.35  5141.0 1619.74
  5148.0 1622.29  5162.2 1624.17  5179.2 1624.37  5219.7 1624.87  5258.3 1625.82
#Mann=8,-1,0
  4639.9    0.16       0  4647.0   0.035       0  4972.6    0.07       0
  5022.1    0.07       0  5062.0    0.07       0  5084.8    0.07       0
  5179.2   0.035       0  5219.7    0.07       0
Bank Sta=5022.1,5062
Exp/Cntr=0.3,0.1

Type RM Length L Ch R = 1,23090,83,83,83
BEGIN DESCRIPTION:
Mapping XS 512d3c43
END DESCRIPTION:
XS GIS Cut Line= 3
      1637138.35      6954065.17      1637135.74      6954540.47
      1637153.97      6954852.93
#Sta/Elev= 30
  4526.9 1613.06  4579.7 1613.36  4589.7 1613.81  4719.7 1613.74  4819.7 1612.21
  4859.7 1611.12  4869.7 1611.25  4899.7 1610.00  4909.7 1609.14  4919.7 1608.14
  4929.7 1606.18  4949.7 1603.50  4959.7 1603.11  4968.3 1602.19  4979.7 1600.71
  4989.6 1598.86  4990.6 1598.36  5029.0 1598.36  5030.0 1598.86  5039.8 1603.16
  5049.8 1604.84  5059.8 1607.35  5069.9 1608.06  5075.1 1609.15  5080.1 1609.10
  5109.9 1616.66  5119.9 1618.14  5125.2 1618.41  5270.2 1621.98  5315.2 1622.54
#Mann=5,-1,0
  4526.9   0.035       0  4968.3    0.07       0  4989.6    0.07       0
  5030.0    0.07       0  5125.2   0.035       0
Bank Sta=4989.6,5030
Exp/Cntr=0.3,0.1

Type RM Length L Ch R = 1,23007,137,137,137
BEGIN DESCRIPTION:
Mapping XS 43da001d
END DESCRIPTION:
XS GIS Cut Line= 4
      1637058.92      6954023.56      1637040.69      6954410.26
      1637052.41      6954541.77      1637058.92      6954852.94
#Sta/Elev= 30
  4484.6 1612.53  4539.1 1612.22  4669.1 1613.19  4759.3 1613.06  4769.4 1612.75
  4799.4 1612.83  4809.4 1612.32  4859.5 1611.76  4868.1 1611.14  4889.5 1610.34
  4899.6 1609.17  4909.6 1608.93  4939.7 1605.21  4949.8 1603.48  4959.8 1602.26
  4980.8 1600.81  4989.7 1597.61  4990.7 1597.11  5029.2 1597.11  5030.2 1597.61
  5040.0 1601.86  5070.0 1608.11  5080.0 1610.59  5100.0 1616.29  5106.2 1616.96
  5130.0 1618.60  5140.0 1618.53  5220.0 1620.23  5270.1 1621.73  5315.0 1622.32
#Mann=4,-1,0
  4484.6   0.035       0  4989.7    0.07       0  5030.2   0.035       0
  5106.2   0.035       0
Bank Sta=4989.7,5030.2
Exp/Cntr=0.3,0.1

Type RM Length L Ch R = 1,22870,395,395,395
BEGIN DESCRIPTION:
Mapping XS 38dbeecf
END DESCRIPTION:
XS GIS Cut Line= 3
      1636888.34      6953988.34      1636915.69      6954539.17
      1636923.46      6954834.56
#Sta/Elev= 30
  4450.9 1611.35  4490.6 1611.44  4510.6 1611.16  4550.7 1611.56  4610.8 1611.22
  4720.9 1612.19  4781.0 1612.38  4841.0 1611.72  4861.1 1611.04  4886.9 1609.02
  4891.9 1609.09  4901.1 1608.03  4921.1 1604.60  4931.1 1604.61  4941.0 1603.34
  4951.2 1600.93  4971.0 1597.37  4972.0 1596.87  5010.5 1596.87  5011.5 1597.37
  5021.2 1601.64  5031.2 1603.04  5061.3 1609.33  5081.3 1615.50  5101.3 1617.22
  5141.3 1618.98  5157.8 1619.18  5161.3 1619.27  5166.3 1618.69  5297.9 1621.21
#Mann=5,-1,0
  4450.9   0.035       0  4941.0    0.07       0  4971.0    0.07       0
  5011.5    0.07       0  5157.8   0.035       0
Bank Sta=4971,5011.5
Exp/Cntr=0.3,0.1

Type RM Length L Ch R = 1,22475,486,486,486
BEGIN DESCRIPTION:
Mapping XS 37ea3657
END DESCRIPTION:
XS GIS Cut Line= 3
      1636537.61      6954039.61      1636553.23      6954440.69
      1636583.05      6954754.39
#Sta/Elev= 30
  4601.7 1608.50  4750.2 1609.19  4840.3 1610.55  4913.8 1608.52  4922.7 1608.45
  4930.3 1607.12  4940.3 1606.07  4956.9 1602.33  4970.4 1599.45  4980.4 1596.31
  4990.2 1594.38  4991.2 1593.88  5029.7 1593.88  5030.7 1594.38  5040.6 1599.50
  5050.6 1601.11  5060.7 1601.90  5070.1 1603.67  5075.2 1603.66  5080.7 1604.53
  5100.8 1608.37  5120.9 1613.88  5151.1 1616.44  5161.1 1616.28  5178.2 1617.11
  5183.3 1616.92  5221.4 1618.16  5261.6 1618.70  5271.6 1619.17  5318.2 1619.09
#Mann=5,-1,0
  4601.7   0.035       0  4913.8    0.07       0  4956.9   0.035       0
  4990.2   0.035       0  5030.7   0.035       0
Bank Sta=4990.2,5030.7
Exp/Cntr=0.3,0.1

Type RM Length L Ch R = 1,21989,492,492,492
BEGIN DESCRIPTION:
Mapping XS 03ff68cc
END DESCRIPTION:
XS GIS Cut Line= 3
      1635880.06      6953979.76      1636084.48      6954391.21
      1636282.39      6954813.06
#Sta/Elev= 30
  4544.4 1615.07  4675.0 1614.05  4697.4 1610.62  4703.0 1607.91  4719.8 1605.48
  4725.4 1603.69  4732.3 1603.40  4837.4 1605.98  4904.6 1604.72  4927.0 1602.22
  4943.8 1598.83  4949.4 1599.53  4955.6 1598.47  4977.9 1598.33  4979.0 1596.88
  4980.0 1596.38  5019.5 1596.88  5022.4 1598.38  5084.9 1599.46  5108.1 1600.04
  5126.3 1602.52  5182.1 1605.02  5199.1 1606.83  5275.2 1607.43  5287.2 1607.51
  5364.6 1608.64  5393.0 1610.44  5415.8 1613.07  5421.3 1614.45  5469.8 1616.13
#Mann=7,-1,0
  4544.4   0.035       0  4979.0   0.035       0  5019.5   0.035       0
  5084.9    0.07       0  5126.3   0.035       0  5275.2    0.07       0
  5287.2   0.035       0
Bank Sta=4979,5019.5
Exp/Cntr=0.3,0.1

Type RM Length L Ch R = 1,21497,464,464,464
BEGIN DESCRIPTION:
Mapping XS 9cf2444d
END DESCRIPTION:
XS GIS Cut Line= 3
      1635457.83      6954369.48      1635702.65      6954645.55
      1636100.52      6954912.10
#Sta/Elev= 30
  4634.6 1609.85  4730.6 1611.91  4737.3 1611.76  4815.9 1612.36  4851.0 1611.86
  4877.6 1610.88  4893.7 1609.15  4900.4 1609.02  4914.6 1607.30  4922.1 1605.54
  4928.8 1604.49  4932.3 1603.39  4943.0 1600.77  4964.8 1591.71  4972.9 1590.93
  4973.9 1590.43  5012.5 1590.43  5013.5 1590.93  5014.7 1593.98  5020.7 1597.79
  5042.5 1599.75  5050.7 1599.67  5065.7 1600.34  5078.6 1601.51  5150.9 1603.59
  5245.8 1605.40  5447.0 1608.04  5462.0 1608.86  5475.9 1610.75  5482.5 1612.07
#Mann=6,-1,0
  4634.6   0.035       0  4737.3    0.07       0  4877.6   0.035       0
  4932.3    0.07       0  4972.9   0.035       0  5013.5   0.035       0
Bank Sta=4972.9,5013.5
Exp/Cntr=0.3,0.1

Type RM Length L Ch R = 1,21033,501,501,501
BEGIN DESCRIPTION:
Mapping XS 2444017e
END DESCRIPTION:
XS GIS Cut Line= 3
      1635016.67      6954510.14      1635303.13      6954848.67
      1635593.91      6955208.89
#Sta/Elev= 30
  4560.6 1610.41  4643.0 1608.64  4649.6 1608.93  4700.2 1607.39  4778.2 1603.68
  4870.5 1602.19  4940.8 1598.37  4962.8 1593.98  4969.3 1593.44  4977.0 1593.78
  4981.3 1592.51  4982.3 1592.01  5021.0 1592.01  5022.0 1592.51  5026.7 1593.85
  5047.5 1596.07  5061.9 1599.95  5068.3 1599.98  5076.3 1601.05  5105.1 1601.54
  5183.1 1601.39  5210.7 1601.75  5225.0 1602.71  5233.0 1604.25  5239.4 1604.55
  5253.8 1608.19  5268.2 1610.38  5289.0 1612.54  5353.0 1614.20  5467.0 1615.82
#Mann=3,-1,0
  4560.6   0.035       0  4981.3   0.035       0  5022.0   0.035       0
Bank Sta=4981.3,5022
Exp/Cntr=0.3,0.1

Type RM Length L Ch R = 1,20532,549,549,549
BEGIN DESCRIPTION:
Mapping XS b086ce77
END DESCRIPTION:
XS GIS Cut Line= 3
      1634738.90      6954563.56      1634860.42      6955032.27
      1635238.02      6955422.89
#Sta/Elev= 30
  4517.9 1608.53  4594.8 1606.88  4641.6 1603.78  4717.6 1601.29  4894.4 1599.15
  4904.7 1598.64  4920.5 1595.05  4935.7 1593.40  4940.7 1591.27  4941.7 1590.77
  4981.4 1591.27  4987.4 1592.29  5023.7 1592.68  5030.6 1593.22  5037.8 1595.25
  5043.3 1595.52  5058.9 1597.87  5080.0 1599.14  5136.6 1599.12  5157.9 1597.96
  5179.0 1598.71  5186.2 1601.11  5193.2 1601.37  5200.4 1604.00  5207.3 1604.47
  5214.5 1606.44  5242.8 1608.72  5263.9 1609.41  5440.9 1608.89  5545.4 1610.84
#Mann=4,-1,0
  4517.9   0.035       0  4940.7    0.07       0  4981.4   0.035       0
  5043.3   0.035       0
Bank Sta=4940.7,4981.4
Exp/Cntr=0.3,0.1

Type RM Length L Ch R = 1,19983,511,511,511
BEGIN DESCRIPTION:
Mapping XS 63bee427
END DESCRIPTION:
XS GIS Cut Line= 3
      1634407.29      6954642.95      1634357.38      6955185.48
      1634359.55      6955448.05
#Sta/Elev= 30
  4460.7 1605.55  4616.4 1602.01  4636.5 1600.73  4645.5 1599.61  4650.5 1599.62
  4656.6 1598.76  4676.7 1597.72  4797.2 1597.67  4827.3 1597.10  4837.3 1594.89
  4847.4 1593.88  4857.4 1595.10  4870.1 1594.88  4927.7 1594.27  4947.8 1592.89
  4955.5 1591.75  4957.8 1591.41  4967.5 1586.43  4968.5 1585.93  5007.5 1585.93
  5008.5 1586.43  5009.3 1591.31  5018.0 1593.44  5028.0 1594.80  5048.0 1598.85
  5058.0 1602.73  5078.0 1605.37  5098.0 1607.19  5178.0 1608.22  5268.1 1608.47
#Mann=5,-1,0
  4460.7   0.035       0  4870.1    0.07       0  4955.5   0.035       0
  4967.5   0.035       0  5008.5   0.035       0
Bank Sta=4967.5,5008.5
Exp/Cntr=0.3,0.1

Type RM Length L Ch R = 1,19472,329,329,329
BEGIN DESCRIPTION:
Mapping XS 196de0dd
END DESCRIPTION:
XS GIS Cut Line= 3
      1634248.86      6954614.75      1633858.25      6955137.74
      1633660.75      6955350.42
#Sta/Elev= 30
  4352.5 1603.60  4443.9 1600.49  4456.8 1599.64  4571.4 1596.42  4615.2 1595.87
  4643.6 1596.19  4671.5 1595.72  4706.9 1595.68  4743.5 1595.81  4786.1 1596.61
  4803.5 1596.23  4893.3 1593.24  4907.0 1591.51  4915.4 1588.68  4930.0 1587.70
  4950.8 1587.77  4965.4 1586.00  4965.7 1585.01  4966.7 1584.51  5005.8 1584.51
  5006.8 1585.01  5008.9 1590.12  5014.9 1592.33  5021.7 1595.97  5029.1 1598.86
  5035.9 1600.86  5043.3 1601.59  5078.4 1602.97  5198.6 1605.62  5295.5 1606.56
#Mann=4,-1,0
  4352.5   0.035       0  4803.5    0.07       0  4965.7   0.035       0
  5006.8   0.035       0
Bank Sta=4965.7,5006.8
Exp/Cntr=0.3,0.1

Type RM Length L Ch R = 1,19143,453,453,453
BEGIN DESCRIPTION:
Mapping XS 78dbbabf
END DESCRIPTION:
XS GIS Cut Line= 3
      1634023.17      6954491.04      1633680.30      6954875.15
      1633485.01      6955087.80
#Sta/Elev= 30
  4493.3 1603.66  4497.0 1603.22  4574.8 1601.16  4617.4 1597.16  4660.0 1595.90
  4716.9 1594.85  4744.5 1595.10  4758.7 1594.58  4794.6 1594.55  4843.9 1593.49
  4879.1 1593.56  4915.0 1594.64  4921.7 1594.49  4927.0 1593.68  4929.2 1593.35
  4947.3 1586.33  4950.1 1585.32  4971.8 1585.31  4972.2 1584.86  4973.2 1584.36
  5012.3 1584.36  5013.3 1584.86  5013.7 1585.60  5027.9 1590.58  5049.5 1593.83
  5063.7 1597.61  5070.5 1600.20  5092.0 1605.13  5162.3 1606.13  5296.9 1606.66
#Mann=5,-1,0
  4493.3   0.035       0  4927.0    0.07       0  4947.3   0.035       0
  4972.2   0.035       0  5013.3   0.035       0
Bank Sta=4972.2,5013.3
Exp/Cntr=0.3,0.1
