--- Chimney Creek 1105.prj (project) ---

Proj Title=Chimney Creek 1105 Base Level Engineering
Current Plan=p01
Default Exp/Contr=0.3,0.1
English Units
Geom File=g01
Flow File=f01
Plan File=p01
BEGIN DESCRIPTION:
Chimney Creek 1105
END DESCRIPTION:

--- Chimney Creek 1105.p01 (plan) ---

Plan Title=Multiple Run
Short Identifier=Multiple
Geom File=g01
Flow File=f01
Subcritical Flow
K Sum by GR= 0
Std Step Tol= 0.01
Critical Tol= 0.01
Num of Std Step Trials= 20
Max Error Tol= 0.3
Flow Tol Ratio= 0.001
Split Flow NTrial= 30
Split Flow Tol= 0.02
Split Flow Ratio= 0.02
Log Output Level= 0
Friction Slope Method= 1
Unsteady Friction Slope Method= 2
Unsteady Bridges Friction Slope Method= 1
Parabolic Critical Depth
Global Vel Dist=  1 , 1 , 1
Global Log Level= 0
CheckData=True
Encroach Param= -1, 0, 0, 0
BEGIN DESCRIPTION:
Multiple Run
END DESCRIPTION:

--- Chimney Creek 1105.f01 (steady flow) ---

Flow Title=Multiple
Number of Profiles=7
Profile Names=10-year,25-year,50-year,1pct_min,100-year,1pct_plu,500-year
River Rch & RM= Chimney Creek 11,Reach-1,18769
     237     327     401     245     489     976     737
River Rch & RM= Chimney Creek 11,Reach-1,17657
     274     382     471     289     577    1151     878
River Rch & RM= Chimney Creek 11,Reach-1,15943
     320     448     555     342     683    1363    1047
River Rch & RM= Chimney Creek 11,Reach-1,12342
     443     628     784     487     971    1937    1509
River Rch & RM= Chimney Creek 11,Reach-1,3850
     529     756     949     592    1181    2357    1854
River Rch & RM= Chimney Creek 11,Reach-1,1394
     600     863    1088     681    1358    2710    2146
Boundary for River Rch & Prof#=Chimney Creek 11,Reach-1,1
Up Type=0
Dn Type=3
Dn Slope=0.005
Boundary for River Rch & Prof#=Chimney Creek 11,Reach-1,2
Up Type=0
Dn Type=3
Dn Slope=0.005
Boundary for River Rch & Prof#=Chimney Creek 11,Reach-1,3
Up Type=0
Dn Type=3
Dn Slope=0.005
Boundary for River Rch & Prof#=Chimney Creek 11,Reach-1,4
Up Type=0
Dn Type=3
Dn Slope=0.005
Boundary for River Rch & Prof#=Chimney Creek 11,Reach-1,5
Up Type=0
Dn Type=3
Dn Slope=0.005
Boundary for River Rch & Prof#=Chimney Creek 11,Reach-1,6
Up Type=0
Dn Type=3
Dn Slope=0.005
Boundary for River Rch & Prof#=Chimney Creek 11,Reach-1,7
Up Type=0
Dn Type=3
Dn Slope=0.005

--- Chimney Creek 1105.g01 (geometry) ---

Geom Title=Existing Conditions

River Reach=Chimney Creek 11,Reach-1
Reach XY= 30
      1643405.00      6946888.00      1642889.79      6946438.51
      1642510.93      6946440.24      1641839.78      6946787.48
      1640956.63      6946641.13      1640461.06      6947129.86
      1639731.53      6947511.01      1639061.05      6948479.84
      1638777.84      6948588.29      1638291.79      6948501.61
      1637307.45      6949682.54      1636865.45      6949786.96
      1636334.95      6949537.40      1635644.56      6949836.94
      1635298.97      6949745.45      1634810.40      6950235.57
      1634903.38      6950581.97      1634658.14      6950796.05
      1634703.81      6951078.41      1634557.44      6951232.53
      1633912.61      6951184.93      1633830.13      6950887.46
      1632570.21      6950938.51      1632202.69      6951093.82
      1632001.45      6951886.53      1631591.38      6952501.24
      1631362.67      6952631.48      1631347.20      6952944.21
      1630708.12      6953339.63      1630955.00      6953838.00

Type RM Length L Ch R = 1,18769,181,181,181
BEGIN DESCRIPTION:
Chimney Creek 1105 28.0
END DESCRIPTION:
XS GIS Cut Line= 3
      1643471.40      6946446.82      1643371.37      6946887.92
      1643276.51      6947224.41
#Sta/Elev= 30
  4547.7 1683.43  4559.2 1683.02  4602.3 1682.46  4630.9 1681.26  4682.2 1680.11
  4688.5 1679.69  4702.7 1679.54  4736.8 1678.38  4774.5 1677.83  4785.0 1677.41
  4795.0 1677.46  4815.5 1676.86  4846.3 1676.69  4877.0 1675.75  4907.8 1675.36
  4919.5 1674.79  4938.6 1674.76  4989.8 1672.33  5003.2 1672.17  5003.4 1671.67
  5006.9 1671.67  5007.2 1672.17  5031.3 1673.39  5044.4 1674.42  5052.0 1675.36
  5124.8 1678.19  5218.3 1680.10  5264.0 1681.54  5322.2 1682.67  5349.6 1682.89
#Mann=3,-1,0
  4547.7   0.035       0  5003.2   0.035       0  5007.2   0.035       0
Bank Sta=5003.2,5007.2
Exp/Cntr=0.3,0.1

Type RM Length L Ch R = 1,18588,63,63,63
BEGIN DESCRIPTION:
Mapping XS 3ea422c1
END DESCRIPTION:
XS GIS Cut Line= 4
      1643406.31      6946509.72      1643306.47      6946733.27
      1643221.84      6946791.86      1643106.93      6947093.23
#Sta/Elev= 30
  4659.3 1681.63  4674.3 1680.80  4690.3 1680.85  4697.5 1680.23  4756.0 1677.99
  4772.6 1677.97  4778.1 1677.44  4842.3 1676.09  4854.5 1674.88  4887.4 1674.92
  4899.7 1673.98  4922.7 1673.27  4937.6 1671.43  4952.4 1668.71  4966.7 1666.99
  4979.5 1666.19  4992.3 1666.12  4992.6 1665.62  4996.1 1665.62  4996.3 1666.12
  5007.1 1666.24  5010.3 1666.72  5015.6 1667.93  5035.0 1671.12  5040.3 1672.71
  5045.7 1673.75  5077.8 1676.31  5110.0 1677.53  5289.7 1681.16  5329.6 1681.64
#Mann=3,-1,0
  4659.3   0.035       0  4992.3   0.035       0  4996.3   0.035       0
Bank Sta=4992.3,4996.3
Exp/Cntr=0.3,0.1

Type RM Length L Ch R = 1,18525,45,45,45
BEGIN DESCRIPTION:
Mapping XS 31dc9cca
END DESCRIPTION:
XS GIS Cut Line= 4
      1643362.89      6946429.47      1643269.58      6946694.21
      1643169.76      6946761.48      1643050.38      6947030.61
#Sta/Elev= 30
  4604.6 1683.77  4687.9 1679.76  4804.5 1676.62  4815.1 1676.05  4825.4 1674.52
  4825.7 1674.02  4829.4 1674.52  4853.1 1674.89  4858.4 1676.13  4868.1 1675.10
  4878.7 1676.97  4884.0 1678.72  4913.9 1678.57  4920.0 1676.72  4934.9 1678.86
  4941.0 1676.97  4949.9 1678.41  4955.9 1675.52  4963.2 1677.88  4976.9 1678.09
  4985.9 1677.25  4991.9 1678.17  4999.4 1677.00  5005.5 1674.94  5012.8 1677.39
  5023.8 1678.12  5035.0 1676.39  5058.2 1675.73  5128.0 1678.20  5300.1 1680.98
#Mann=3,-1,0
  4604.6   0.035       0  4825.4   0.035       0  4829.4   0.035       0
Bank Sta=4825.4,4829.4
Exp/Cntr=0.3,0.1

Type RM Length L Ch R = 1,18480,328,328,328
BEGIN DESCRIPTION:
Mapping XS 17577db0
END DESCRIPTION:
XS GIS Cut Line= 4
      1643297.80      6946386.04      1643217.50      6946644.29
      1643152.39      6946722.42      1642967.94      6947013.21
#Sta/Elev= 30
  4632.5 1683.32  4686.9 1681.25  4707.9 1679.87  4730.1 1679.06  4795.2 1677.32
  4802.1 1676.72  4822.5 1676.48  4833.5 1675.72  4854.5 1675.44  4875.4 1673.17
  4885.9 1674.54  4902.3 1672.42  4969.7 1670.19  4970.0 1669.69  4973.5 1669.69
  4973.7 1670.19  4992.6 1671.11  5004.6 1670.79  5022.5 1671.28  5028.4 1670.82
  5043.7 1671.97  5049.6 1672.02  5058.6 1674.69  5064.8 1675.17  5094.1 1676.61
  5129.7 1677.78  5165.2 1678.56  5295.5 1680.27  5319.1 1680.39  5349.0 1679.88
#Mann=3,-1,0
  4632.5   0.035       0  4969.7   0.035       0  4973.7   0.035       0
Bank Sta=4969.7,4973.7
Exp/Cntr=0.3,0.1

Type RM Length L Ch R = 1,18152,249,249,249
BEGIN DESCRIPTION:
Mapping XS 71bd5986
END DESCRIPTION:
XS GIS Cut Line= 3
      1643020.86      6946201.69      1642960.08      6946486.45
      1642913.35      6946924.39
#Sta/Elev= 30
  4710.3 1684.06  4718.1 1683.10  4727.0 1683.49  4737.2 1682.65  4756.1 1682.08
  4788.3 1680.10  4812.1 1679.12  4819.0 1678.39  4849.7 1677.04  4880.4 1675.00
  4890.6 1674.94  4900.8 1674.32  4911.1 1673.12  4941.7 1670.97  4962.2 1668.33
  4980.6 1667.24  4980.9 1666.74  4984.4 1666.74  4984.6 1667.24  5005.2 1668.18
  5023.1 1669.94  5063.4 1671.40  5097.5 1671.94  5174.0 1673.92  5224.3 1676.32
  5264.5 1676.77  5282.3 1677.72  5287.3 1677.60  5304.7 1678.36  5441.9 1678.59
#Mann=4,-1,0
  4710.3    0.07       0  4756.1   0.035       0  4980.6   0.035       0
  4984.6   0.035       0
Bank Sta=4980.6,4984.6
Exp/Cntr=0.3,0.1

Type RM Length L Ch R = 1,17903,246,246,246
BEGIN DESCRIPTION:
Mapping XS 4f12570f
END DESCRIPTION:
XS GIS Cut Line= 3
      1642843.77      6946123.60      1642725.71      6946441.31
      1642630.23      6947048.91
#Sta/Elev= 30
  4664.6 1681.72  4700.0 1681.07  4705.4 1680.55  4744.0 1680.18  4780.3 1678.45
  4829.3 1676.00  4846.5 1674.64  4907.2 1671.87  4962.6 1668.25  4968.0 1667.40
  4997.1 1666.31  4997.4 1665.81  5000.9 1665.81  5001.1 1666.31  5008.8 1666.42
  5030.6 1667.12  5038.0 1668.07  5071.0 1669.91  5111.5 1670.93  5168.2 1671.97
  5230.8 1672.65  5235.8 1672.27  5303.9 1673.34  5361.0 1675.41  5374.7 1675.38
  5455.7 1677.74  5496.3 1679.45  5536.7 1679.33  5597.4 1679.98  5618.6 1681.06
#Mann=5,-1,0
  4664.6   0.035       0  4780.3    0.07       0  4997.1    0.07       0
  5001.1    0.07       0  5008.8   0.035       0
Bank Sta=4997.1,5001.1
Exp/Cntr=0.3,0.1

Type RM Length L Ch R = 1,17657,280,280,280
BEGIN DESCRIPTION:
Mapping XS 43525a76
END DESCRIPTION:
XS GIS Cut Line= 3
      1642364.94      6946131.24      1642486.47      6946457.63
      1642554.18      6947009.71
#Sta/Elev= 30
  4652.5 1681.28  4776.7 1677.60  4787.8 1676.49  4807.0 1676.04  4873.1 1671.44
  4894.7 1670.46  4923.0 1669.19  4928.4 1667.71  4937.2 1666.17  4953.4 1664.70
  4958.7 1665.28  4969.2 1665.37  5009.1 1664.51  5009.4 1664.01  5013.1 1664.01
  5013.4 1664.51  5021.3 1664.76  5041.4 1666.79  5071.7 1668.09  5109.4 1668.67
  5142.2 1670.12  5166.6 1670.42  5283.3 1674.27  5293.3 1674.18  5394.1 1677.03
  5424.3 1677.45  5440.0 1678.52  5464.6 1678.41  5535.1 1680.09  5557.0 1681.10
#Mann=6,-1,0
  4652.5    0.07       0  4894.7   0.035       0  5009.1   0.035       0
  5013.4   0.035       0  5041.4    0.07       0  5166.6   0.035       0
Bank Sta=5009.1,5013.4
Exp/Cntr=0.3,0.1

Type RM Length L Ch R = 1,17377,374,374,374
BEGIN DESCRIPTION:
Mapping XS 39332279
END DESCRIPTION:
XS GIS Cut Line= 3
      1642169.95      6946267.81      1642254.59      6946593.34
      1642328.80      6946907.13
#Sta/Elev= 30
  4664.0 1679.06  4666.8 1679.21  4702.1 1677.65  4707.3 1677.81  4777.9 1676.11
  4783.2 1675.51  4823.8 1674.19  4829.5 1673.60  4870.8 1671.36  4891.5 1670.76
  4945.6 1668.05  4974.2 1665.93  4985.9 1664.03  4994.8 1663.15  5000.2 1662.01
  5011.6 1661.86  5013.3 1661.82  5013.6 1661.32  5017.3 1661.32  5017.6 1661.82
  5036.0 1662.49  5054.0 1664.08  5111.9 1667.57  5149.0 1669.11  5159.3 1670.29
  5201.6 1671.71  5231.2 1673.26  5286.1 1675.07  5303.1 1676.20  5322.8 1676.76
#Mann=6,-1,0
  4664.0    0.07       0  4945.6   0.035       0  5011.6    0.07       0
  5013.3   0.035       0  5017.6    0.07       0  5054.0   0.035       0
Bank Sta=5013.3,5017.6
Exp/Cntr=0.3,0.1

Type RM Length L Ch R = 1,17003,352,352,352
BEGIN DESCRIPTION:
Mapping XS a8229e00
END DESCRIPTION:
XS GIS Cut Line= 3
      1641936.88      6946261.34      1641936.88      6946741.78
      1641916.05      6947118.07
#Sta/Elev= 30
  4523.7 1675.12  4530.4 1674.60  4560.4 1673.77  4631.3 1672.62  4700.4 1671.44
  4720.4 1670.62  4760.4 1670.03  4820.4 1668.36  4853.3 1667.00  4890.4 1665.34
  4970.4 1663.46  5003.0 1661.80  5010.4 1660.94  5028.2 1660.29  5028.5 1659.79
  5032.2 1659.79  5032.5 1660.29  5040.4 1661.87  5050.4 1664.32  5070.5 1666.02
  5127.1 1668.97  5132.1 1668.55  5140.6 1669.33  5150.6 1669.67  5180.6 1671.56
  5212.1 1672.42  5280.8 1674.74  5330.9 1675.78  5360.9 1676.89  5381.0 1677.08
#Mann=7,-1,0
  4523.7   0.035       0  4631.3    0.07       0  4853.3   0.035       0
  5003.0    0.07       0  5028.2   0.035       0  5032.5    0.07       0
  5212.1   0.035       0
Bank Sta=5028.2,5032.5
Exp/Cntr=0.3,0.1

Type RM Length L Ch R = 1,16651,323,323,323
BEGIN DESCRIPTION:
Mapping XS 4e2e36bf
END DESCRIPTION:
XS GIS Cut Line= 3
      1641640.25      6946391.50      1641601.19      6946790.79
      1641590.00      6947013.01
#Sta/Elev= 30
  4601.2 1673.47  4603.3 1672.99  4617.8 1672.63  4627.8 1671.96  4672.2 1670.57
  4713.2 1668.59  4738.3 1667.93  4778.5 1666.23  4798.6 1665.51  4811.5 1665.37
  4828.8 1664.55  4899.1 1662.84  4929.3 1661.38  4939.3 1661.36  4959.4 1660.56
  4975.3 1659.42  4987.3 1658.83  4987.6 1658.33  4991.4 1658.33  4991.7 1658.83
  5002.4 1658.88  5009.6 1659.32  5019.6 1661.48  5025.4 1663.74  5049.7 1664.92
  5094.2 1667.76  5119.8 1668.74  5129.8 1668.77  5149.8 1670.32  5224.9 1672.39
#Mann=7,-1,0
  4601.2   0.035       0  4672.2    0.07       0  4713.2   0.035       0
  4975.3    0.07       0  4987.3    0.07       0  4991.7    0.07       0
  5094.2   0.035       0
Bank Sta=4987.3,4991.7
Exp/Cntr=0.3,0.1

Type RM Length L Ch R = 1,16328,385,385,385
BEGIN DESCRIPTION:
Mapping XS fff12c2e
END DESCRIPTION:
XS GIS Cut Line= 3
      1641356.00      6946440.80      1641293.50      6946741.57
      1641287.01      6946973.78
#Sta/Elev= 30
  4696.0 1669.66  4727.2 1667.90  4764.6 1664.57  4805.5 1662.85  4846.3 1660.32
  4866.8 1659.99  4877.5 1658.85  4887.2 1658.36  4922.5 1657.94  4948.5 1659.02
  4972.6 1658.60  4987.1 1657.54  4987.4 1657.04  4991.2 1657.04  4991.5 1657.54
  5003.2 1657.72  5009.6 1658.25  5019.6 1659.70  5029.6 1661.80  5069.7 1664.40
  5089.7 1664.56  5119.7 1665.52  5126.6 1666.12  5131.6 1665.78  5139.7 1666.49
  5169.7 1666.92  5189.7 1667.57  5199.7 1668.36  5209.7 1668.04  5235.5 1669.39
#Mann=3,-1,0
  4696.0   0.035       0  4987.1   0.035       0  4991.5   0.035       0
Bank Sta=4987.1,4991.5
Exp/Cntr=0.3,0.1

Type RM Length L Ch R = 1,15943,438,438,438
BEGIN DESCRIPTION:
Mapping XS 25dd3b95
END DESCRIPTION:
XS GIS Cut Line= 3
      1640789.61      6946443.42      1640944.54      6946649.12
      1641110.01      6947033.06
#Sta/Elev= 30
  4742.7 1670.97  4749.0 1670.49  4778.2 1670.21  4836.1 1668.18  4849.0 1667.44
  4879.9 1664.67  4898.9 1661.43  4921.8 1659.33  4936.2 1657.48  4957.2 1655.93
  4978.0 1655.11  4996.4 1653.77  5006.8 1653.69  5007.1 1653.19  5011.3 1653.19
  5011.7 1653.69  5031.7 1653.88  5053.4 1655.44  5066.4 1656.77  5097.0 1658.52
  5151.4 1660.36  5184.1 1661.00  5195.7 1661.87  5213.7 1661.83  5227.7 1662.63
  5237.3 1662.50  5266.2 1663.54  5289.8 1663.47  5380.1 1665.73  5418.3 1666.12
#Mann=5,-1,0
  4742.7   0.035       0  4879.9    0.07       0  5006.8    0.07       0
  5011.7    0.07       0  5066.4   0.035       0
Bank Sta=5006.8,5011.7
Exp/Cntr=0.3,0.1

Type RM Length L Ch R = 1,15505,71,71,71
BEGIN DESCRIPTION:
Mapping XS fd0aab95
END DESCRIPTION:
XS GIS Cut Line= 4
      1640507.04      6946606.17      1640525.27      6946766.31
      1640646.36      6946948.60      1640904.15      6947219.40
#Sta/Elev= 30
  4620.2 1670.95  4725.3 1667.82  4846.8 1663.10  4861.8 1660.78  4918.9 1656.29
  4949.0 1651.63  4955.0 1649.78  4970.1 1650.81  4976.1 1648.81  4985.1 1650.41
  4991.1 1648.18  4996.9 1650.12  5002.9 1650.12  5005.9 1647.69  5013.1 1649.50
  5017.6 1647.29  5017.9 1646.79  5022.5 1647.29  5034.2 1651.98  5041.1 1650.43
  5044.1 1651.16  5048.4 1652.21  5055.3 1651.02  5062.5 1652.72  5069.4 1651.93
  5097.7 1653.30  5132.3 1656.98  5189.9 1662.47  5368.8 1666.06  5374.1 1666.21
#Mann=7,-1,0
  4620.2   0.035       0  4725.3    0.07       0  5017.6    0.07       0
  5022.5    0.07       0  5044.1   0.035       0  5132.3    0.07       0
  5368.8   0.035       0
Bank Sta=5017.6,5022.5
Exp/Cntr=0.3,0.1

Type RM Length L Ch R = 1,15434,53,53,53
BEGIN DESCRIPTION:
Mapping XS 32264fc0
END DESCRIPTION:
XS GIS Cut Line= 3
      1640358.58      6946718.11      1640596.88      6946999.38
      1640797.42      6947292.38
#Sta/Elev= 30
  4633.8 1668.83  4664.6 1667.96  4830.3 1662.82  4837.0 1665.00  4843.5 1664.90
  4851.2 1666.83  4865.5 1662.20  4872.1 1664.58  4879.8 1661.74  4886.4 1665.82
  4894.1 1663.38  4900.7 1665.71  4908.4 1664.54  4914.9 1666.34  4929.2 1665.35
  4964.4 1665.44  4972.1 1666.40  4992.9 1664.53  5007.4 1666.14  5028.4 1665.27
  5043.3 1666.45  5079.2 1665.71  5144.9 1667.03  5158.3 1665.25  5165.8 1662.09
  5178.3 1660.98  5178.6 1660.48  5183.2 1660.98  5319.1 1664.88  5357.5 1665.21
#Mann=5,-1,0
  4633.8   0.035       0  4664.6    0.07       0  5178.3    0.07       0
  5183.2    0.07       0  5319.1   0.035       0
Bank Sta=5178.3,5183.2
Exp/Cntr=0.3,0.1

Type RM Length L Ch R = 1,15381,618,618,618
BEGIN DESCRIPTION:
Mapping XS 78956871
END DESCRIPTION:
XS GIS Cut Line= 6
      1640195.84      6946783.23      1640425.01      6946876.98
      1640534.38      6947007.19      1640557.82      6947035.84
      1640599.49      6947106.15      1640669.75      6947383.28
#Sta/Elev= 30
  4545.8 1666.10  4649.2 1665.95  4717.8 1664.33  4780.0 1663.58  4797.3 1663.16
  4836.4 1661.12  4844.1 1660.32  4865.0 1659.34  4872.7 1658.20  4907.9 1655.69
  4928.7 1656.35  4950.8 1655.63  4957.3 1656.08  4960.7 1655.46  4971.6 1654.97
  5006.8 1655.50  5041.4 1654.37  5041.7 1653.87  5045.9 1653.87  5046.3 1654.37
  5059.4 1655.11  5065.3 1655.96  5072.7 1655.67  5080.4 1656.04  5094.4 1657.35
  5135.7 1658.00  5146.0 1659.24  5168.7 1660.85  5215.9 1661.57  5368.1 1665.09
#Mann=4,-1,0
  4545.8    0.07       0  5041.4    0.07       0  5046.3    0.07       0
  5215.9   0.035       0
Bank Sta=5041.4,5046.3
Exp/Cntr=0.3,0.1

Type RM Length L Ch R = 1,14763,156,156,156
BEGIN DESCRIPTION:
Mapping XS 9126c9d5
END DESCRIPTION:
XS GIS Cut Line= 3
      1640013.55      6946961.32      1640043.06      6947341.48
      1640119.45      6947950.81
#Sta/Elev= 30
  4623.6 1664.95  4700.5 1662.76  4706.2 1662.23  4754.5 1660.51  4810.8 1658.31
  4823.7 1657.55  4851.0 1655.65  4881.1 1652.88  4901.1 1651.46  4921.2 1650.51
  4941.2 1648.91  4978.9 1647.94  4979.2 1647.44  4983.5 1647.44  4983.9 1647.94
  5021.6 1648.28  5031.6 1649.02  5041.7 1649.24  5071.9 1650.97  5144.3 1653.01
  5219.8 1654.03  5224.8 1654.42  5263.4 1655.38  5283.6 1655.38  5385.8 1657.14
  5461.3 1657.94  5466.3 1658.27  5515.4 1659.12  5525.5 1658.98  5619.0 1659.97
#Mann=5,-1,0
  4623.6   0.035       0  4754.5    0.07       0  4823.7   0.035       0
  4978.9   0.035       0  4983.9   0.035       0
Bank Sta=4978.9,4983.9
Exp/Cntr=0.3,0.1

Type RM Length L Ch R = 1,14607,261,261,261
BEGIN DESCRIPTION:
Mapping XS 8c1c0d4f
END DESCRIPTION:
XS GIS Cut Line= 3
      1639864.59      6947040.92      1639902.79      6947396.86
      1639979.17      6947957.59
#Sta/Elev= 30
  4644.9 1662.27  4696.5 1661.20  4788.6 1657.73  4823.0 1657.05  4843.1 1655.65
  4880.7 1653.83  4893.4 1653.73  4913.5 1652.55  4933.6 1650.64  4953.7 1647.84
  4970.3 1647.22  4970.7 1646.72  4975.0 1646.72  4975.3 1647.22  4994.0 1647.67
  5024.2 1647.55  5057.9 1649.02  5125.1 1649.15  5165.5 1651.11  5266.4 1653.41
  5275.0 1653.25  5280.1 1653.62  5327.0 1654.21  5347.2 1653.96  5352.5 1654.58
  5407.7 1654.93  5458.2 1655.85  5497.2 1655.59  5508.7 1656.19  5568.8 1656.79
#Mann=3,-1,0
  4644.9   0.035       0  4970.3   0.035       0  4975.3   0.035       0
Bank Sta=4970.3,4975.3
Exp/Cntr=0.3,0.1

Type RM Length L Ch R = 1,14346,334,334,334
BEGIN DESCRIPTION:
Mapping XS 9f1f5b3f
END DESCRIPTION:
XS GIS Cut Line= 3
      1639598.34      6947310.92      1639700.77      6947548.76
      1639844.86      6947977.54
#Sta/Elev= 30
  4746.2 1654.68  4773.0 1654.42  4786.6 1654.75  4796.5 1654.16  4854.4 1653.39
  4862.8 1653.58  4878.0 1652.64  4895.5 1652.52  4925.0 1651.50  4948.5 1650.03
  4971.7 1646.90  4977.5 1645.74  4993.4 1644.50  5001.0 1644.71  5001.7 1644.26
  5002.0 1643.76  5006.3 1643.76  5006.7 1644.26  5025.5 1644.90  5037.7 1646.13
  5141.5 1648.52  5152.1 1648.50  5173.1 1649.27  5183.7 1649.23  5258.4 1651.78
  5284.6 1651.90  5373.6 1653.40  5394.7 1653.52  5410.7 1653.20  5457.5 1654.23
#Mann=3,-1,0
  4746.2   0.035       0  5001.7   0.035       0  5006.7   0.035       0
Bank Sta=5001.7,5006.7
Exp/Cntr=0.3,0.1

Type RM Length L Ch R = 1,14012,383,383,383
BEGIN DESCRIPTION:
Mapping XS 514c333d
END DESCRIPTION:
XS GIS Cut Line= 3
      1639339.44      6947635.85      1639495.69      6947799.70
      1639773.10      6948133.45
#Sta/Elev= 30
  4775.6 1651.27  4802.3 1651.39  4809.3 1651.00  4908.3 1650.00  4958.0 1647.95
  4979.1 1645.60  4986.0 1643.99  4993.3 1643.37  5004.2 1643.25  5005.0 1642.70
  5005.4 1642.20  5009.7 1642.20  5010.1 1642.70  5014.0 1643.14  5036.2 1643.39
  5057.0 1645.12  5085.6 1645.44  5106.5 1646.45  5149.4 1647.40  5184.6 1649.01
  5206.7 1649.29  5213.2 1650.11  5227.6 1649.77  5248.4 1650.85  5256.2 1650.67
  5262.7 1651.24  5305.7 1651.82  5320.0 1652.45  5376.9 1653.02  5436.0 1654.44
#Mann=3,-1,0
  4775.6   0.035       0  5005.0   0.035       0  5010.1   0.035       0
Bank Sta=5005,5010.1
Exp/Cntr=0.3,0.1

Type RM Length L Ch R = 1,13629,431,431,431
BEGIN DESCRIPTION:
Mapping XS 3e540148
END DESCRIPTION:
XS GIS Cut Line= 3
      1639181.15      6947979.85      1639360.15      6948136.07
      1639575.02      6948321.64
#Sta/Elev= 30
  4761.6 1647.90  4833.5 1647.11  4841.1 1646.57  4883.8 1645.71  4918.9 1644.33
  4939.8 1642.94  4990.1 1643.01  4999.1 1642.39  5004.5 1642.39  5011.0 1641.63
  5022.7 1641.00  5023.1 1640.50  5027.4 1640.50  5027.8 1641.00  5032.0 1641.89
  5046.1 1643.03  5053.8 1644.30  5068.0 1645.25  5103.1 1646.40  5124.5 1647.68
  5138.3 1647.69  5145.9 1648.37  5152.5 1648.35  5160.2 1648.95  5166.8 1648.86
  5195.3 1649.67  5244.7 1651.47  5252.3 1651.33  5273.2 1651.98  5283.1 1651.94
#Mann=3,-1,0
  4761.6   0.035       0  5022.7   0.035       0  5027.8   0.035       0
Bank Sta=5022.7,5027.8
Exp/Cntr=0.3,0.1

Type RM Length L Ch R = 1,13198,423,423,423
BEGIN DESCRIPTION:
Mapping XS e6be4aaa
END DESCRIPTION:
XS GIS Cut Line= 3
      1639042.22      6948121.96      1639096.48      6948447.48
      1639133.37      6948662.32
#Sta/Elev= 30
  4670.6 1645.99  4697.0 1645.41  4707.1 1645.62  4747.7 1645.11  4768.0 1645.10
  4775.9 1644.67  4788.2 1644.51  4818.7 1644.47  4836.7 1643.69  4849.1 1643.65
  4859.2 1643.24  4940.3 1642.25  4963.4 1641.00  4978.3 1638.86  4978.7 1638.36
  4983.0 1638.36  4983.4 1638.86  5003.4 1639.15  5011.3 1640.01  5018.9 1641.15
  5024.0 1642.23  5031.6 1643.29  5051.9 1644.09  5072.2 1644.59  5092.5 1645.55
  5138.9 1646.49  5143.9 1646.83  5198.8 1647.07  5204.1 1647.32  5218.6 1647.24
#Mann=3,-1,0
  4670.6   0.035       0  4978.3   0.035       0  4983.4   0.035       0
Bank Sta=4978.3,4983.4
Exp/Cntr=0.3,0.1

Type RM Length L Ch R = 1,12775,433,433,433
BEGIN DESCRIPTION:
Mapping XS 74ddc5f7
END DESCRIPTION:
XS GIS Cut Line= 3
      1638750.56      6948249.74      1638719.09      6948590.50
      1638770.05      6948909.24
#Sta/Elev= 30
  4660.1 1642.52  4678.4 1642.19  4688.5 1642.38  4748.7 1642.02  4758.8 1641.28
  4768.8 1641.78  4929.5 1640.37  4949.6 1639.80  4979.7 1637.72  4986.0 1636.98
  4986.4 1636.48  4990.8 1636.48  4991.1 1636.98  5002.3 1637.02  5006.5 1637.83
  5011.5 1637.84  5020.0 1639.77  5030.2 1641.14  5060.5 1642.37  5068.5 1642.46
  5073.6 1642.92  5130.6 1643.57  5135.6 1643.32  5171.9 1643.54  5192.2 1643.35
  5202.7 1643.65  5242.8 1643.73  5253.0 1643.36  5273.2 1643.81  5325.1 1643.40
#Mann=3,-1,0
  4660.1   0.035       0  4986.0   0.035       0  4991.1   0.035       0
Bank Sta=4986,4991.1
Exp/Cntr=0.3,0.1

Type RM Length L Ch R = 1,12342,450,450,450
BEGIN DESCRIPTION:
Mapping XS e22e29c2
END DESCRIPTION:
XS GIS Cut Line= 3
      1638249.26      6948258.47      1638359.93      6948480.90
      1638582.30      6948803.06
#Sta/Elev= 30
  4752.4 1647.68  4830.1 1643.91  4865.4 1642.68  4890.1 1641.01  4929.3 1639.45
  4951.7 1638.06  4957.3 1637.65  4964.1 1636.22  4971.2 1635.51  4971.7 1635.01
  4976.5 1635.01  4977.0 1635.51  4979.7 1636.10  4986.4 1636.50  5000.9 1636.62
  5017.1 1637.68  5031.9 1637.95  5045.9 1638.01  5073.8 1637.47  5109.7 1637.78
  5124.6 1638.17  5139.4 1639.01  5181.3 1639.51  5203.9 1640.20  5240.3 1640.36
  5267.9 1641.08  5276.7 1640.86  5312.5 1641.54  5369.3 1641.65  5392.3 1642.14
#Mann=4,-1,0
  4752.4    0.07       0  4865.4   0.035       0  4971.2   0.035       0
  4977.0   0.035       0
Bank Sta=4971.2,4977
Exp/Cntr=0.3,0.1

Type RM Length L Ch R = 1,11892,473,473,473
BEGIN DESCRIPTION:
Mapping XS bdef1adc
END DESCRIPTION:
XS GIS Cut Line= 3
      1637892.97      6948290.03      1638025.34      6948769.59
      1638489.75      6949125.50
#Sta/Elev= 30
  4504.1 1644.99  4563.6 1644.11  4568.8 1644.48  4603.1 1643.38  4607.2 1643.65
  4642.7 1642.45  4823.6 1640.84  4844.3 1639.89  4869.5 1637.01  4909.1 1636.94
  4943.4 1636.29  4968.8 1633.56  4982.9 1633.35  4986.7 1632.74  4987.1 1632.24
  4992.0 1632.24  4992.5 1632.74  5007.3 1632.82  5021.9 1634.31  5064.2 1635.87
  5107.0 1636.00  5121.6 1636.57  5156.9 1636.48  5165.0 1637.01  5171.4 1636.69
  5215.0 1637.08  5385.4 1639.09  5555.8 1639.95  5564.0 1640.49  5586.7 1640.04
#Mann=4,-1,0
  4504.1    0.07       0  4607.2   0.035       0  4986.7   0.035       0
  4992.5   0.035       0
Bank Sta=4986.7,4992.5
Exp/Cntr=0.3,0.1

Type RM Length L Ch R = 1,11419,624,624,624
BEGIN DESCRIPTION:
Mapping XS b65cd89d
END DESCRIPTION:
XS GIS Cut Line= 3
      1637275.47      6948744.43      1637752.88      6949137.22
      1638420.65      6949668.40
#Sta/Elev= 30
  4384.2 1647.27  4478.5 1642.50  4492.9 1642.49  4500.1 1641.89  4542.4 1640.34
  4634.9 1637.64  4826.5 1633.90  4947.7 1633.29  4968.6 1632.82  4997.2 1631.68
  4997.5 1631.34  4998.0 1630.84  5003.2 1630.84  5003.7 1631.34  5026.0 1631.75
  5040.5 1633.04  5160.6 1635.14  5367.2 1636.28  5410.5 1636.34  5424.9 1635.73
  5439.3 1636.39  5503.4 1636.52  5666.8 1638.62  5722.8 1638.90  5745.3 1639.55
  5772.5 1639.31  5822.9 1640.04  5830.1 1639.49  5836.5 1640.14  5855.7 1640.33
#Mann=3,-1,0
  4384.2   0.035       0  4997.5   0.035       0  5003.7   0.035       0
Bank Sta=4997.5,5003.7
Exp/Cntr=0.3,0.1

Type RM Length L Ch R = 1,10795,512,512,512
BEGIN DESCRIPTION:
Mapping XS 50e8a494
END DESCRIPTION:
XS GIS Cut Line= 3
      1637110.22      6949070.27      1637375.83      6949615.37
      1637669.24      6950196.99
#Sta/Elev= 30
  4392.2 1645.25  4463.0 1640.02  4478.8 1637.98  4512.0 1634.95  4589.9 1632.18
  4641.4 1628.71  4656.6 1628.39  4663.9 1629.05  4669.5 1628.68  4745.6 1630.97
  4901.4 1631.69  4934.4 1629.45  4945.9 1627.86  4953.5 1627.75  4954.0 1627.25
  4959.9 1627.25  4960.4 1627.75  4985.0 1629.36  5013.1 1629.74  5046.3 1631.43
  5124.7 1632.88  5247.2 1633.41  5252.8 1633.98  5259.1 1633.23  5275.1 1634.07
  5291.8 1633.52  5425.6 1634.45  5438.3 1633.98  5470.2 1634.73  5650.0 1635.01
#Mann=5,-1,0
  4392.2   0.035       0  4463.0    0.07       0  4478.8   0.035       0
  4953.5   0.035       0  4960.4   0.035       0
Bank Sta=4953.5,4960.4
Exp/Cntr=0.3,0.1

Type RM Length L Ch R = 1,10283,139,139,139
BEGIN DESCRIPTION:
Mapping XS 59bba16c
END DESCRIPTION:
XS GIS Cut Line= 3
      1636977.61      6949184.85      1636950.26      6949791.59
      1636955.77      6950013.76
#Sta/Elev= 30
  4395.6 1641.16  4413.8 1640.52  4428.8 1639.90  4438.8 1638.39  4458.8 1633.32
  4478.8 1630.71  4488.8 1630.21  4548.9 1630.06  4558.9 1629.67  4564.2 1628.40
  4569.3 1628.63  4578.9 1626.90  4619.0 1626.67  4629.0 1627.43  4639.0 1629.75
  4649.0 1630.11  4809.2 1627.98  4869.2 1629.09  4929.3 1629.31  4979.3 1628.11
  4989.4 1626.93  4995.2 1625.37  4995.7 1624.87  5001.6 1624.87  5002.1 1625.37
  5019.4 1627.10  5029.4 1629.12  5039.4 1629.48  5099.4 1629.98  5225.2 1629.75
#Mann=4,-1,0
  4395.6    0.07       0  4413.8   0.035       0  4995.2   0.035       0
  5002.1   0.035       0
Bank Sta=4995.2,5002.1
Exp/Cntr=0.3,0.1

Type RM Length L Ch R = 1,10144,440,440,440
BEGIN DESCRIPTION:
Mapping XS 1dd1a3f4
END DESCRIPTION:
XS GIS Cut Line= 3
      1636803.13      6949218.66      1636822.66      6949757.73
      1636828.63      6950032.45
#Sta/Elev= 30
  4462.2 1640.38  4481.5 1639.12  4491.6 1638.04  4501.6 1636.12  4524.6 1633.79
  4591.6 1629.48  4611.6 1628.72  4621.6 1629.13  4641.7 1629.00  4654.3 1626.72
  4661.7 1626.32  4691.7 1626.45  4701.7 1627.11  4711.7 1628.47  4771.7 1629.36
  4851.8 1628.94  4881.8 1627.32  4901.8 1626.95  4932.5 1627.90  4961.9 1627.86
  4971.9 1627.33  4991.9 1627.10  4999.3 1626.19  5018.4 1625.87  5018.9 1625.37
  5024.8 1625.37  5025.3 1625.87  5061.9 1629.19  5091.9 1629.67  5276.4 1629.47
#Mann=4,-1,0
  4462.2    0.07       0  4524.6   0.035       0  5018.4   0.035       0
  5025.3   0.035       0
Bank Sta=5018.4,5025.3
Exp/Cntr=0.3,0.1

Type RM Length L Ch R = 1,9704,748,748,748
BEGIN DESCRIPTION:
Mapping XS 235fcf4a
END DESCRIPTION:
XS GIS Cut Line= 3
      1636497.71      6949020.09      1636465.89      6949589.76
      1636556.30      6950780.07
#Sta/Elev= 30
  4433.1 1644.60  4521.1 1644.18  4591.3 1642.68  4651.4 1640.33  4721.3 1635.56
  4761.5 1630.72  4791.6 1629.28  4871.7 1627.20  4951.8 1626.83  4971.8 1625.63
  5028.5 1623.77  5029.0 1623.27  5035.0 1623.27  5035.5 1623.77  5042.0 1624.16
  5052.0 1626.16  5132.3 1627.44  5172.4 1627.13  5393.0 1628.20  5413.1 1627.67
  5483.3 1628.33  5814.2 1628.48  5849.7 1627.85  5864.4 1628.42  5874.4 1628.01
  5934.6 1628.23  5954.6 1627.64  5985.9 1628.11  6085.0 1627.58  6197.4 1627.82
#Mann=4,-1,0
  4433.1    0.07       0  4721.3   0.035       0  5028.5   0.035       0
  5035.5   0.035       0
Bank Sta=5028.5,5035.5
Exp/Cntr=0.3,0.1

Type RM Length L Ch R = 1,8956,337,337,337
BEGIN DESCRIPTION:
Mapping XS d533310c
END DESCRIPTION:
XS GIS Cut Line= 3
      1635870.65      6949341.78      1635801.65      6949742.79
      1635797.74      6950178.97
#Sta/Elev= 30
  4598.0 1628.89  4600.5 1628.56  4614.5 1628.33  4644.9 1628.30  4685.5 1627.50
  4720.4 1627.26  4726.1 1626.79  4780.3 1626.22  4787.0 1625.84  4817.4 1625.72
  4835.2 1625.07  4888.4 1624.64  4929.0 1623.41  4939.2 1622.14  4949.3 1621.80
  5006.6 1620.77  5007.1 1620.27  5013.1 1620.27  5013.6 1620.77  5040.1 1623.54
  5050.1 1624.10  5090.1 1624.61  5120.1 1624.26  5160.1 1624.52  5200.1 1624.19
  5220.1 1624.72  5250.1 1624.91  5400.1 1625.21  5420.1 1624.98  5441.1 1625.26
#Mann=3,-1,0
  4598.0   0.035       0  5006.6   0.035       0  5013.6   0.035       0
Bank Sta=5006.6,5013.6
Exp/Cntr=0.3,0.1

Type RM Length L Ch R = 1,8619,400,400,400
BEGIN DESCRIPTION:
Mapping XS 35ea16b7
END DESCRIPTION:
XS GIS Cut Line= 3
      1635388.87      6949452.39      1635502.17      6949836.54
      1635801.87      6950793.71
#Sta/Elev= 30
  4597.8 1631.84  4600.1 1631.23  4633.4 1630.40  4638.6 1629.67  4699.6 1626.94
  4760.0 1624.61  4770.5 1623.33  4782.3 1620.53  4810.4 1621.55  4864.3 1621.17
  4887.5 1622.43  4987.4 1622.71  4996.5 1621.65  5001.7 1621.65  5021.8 1619.07
  5022.3 1618.57  5028.3 1618.57  5028.8 1619.07  5031.3 1620.21  5052.2 1622.87
  5083.7 1623.63  5160.3 1623.13  5502.8 1624.15  5607.6 1623.75  5830.3 1623.81
  5857.5 1624.23  5869.6 1623.72  5911.5 1624.23  5932.9 1623.55  6001.3 1624.02
#Mann=4,-1,0
  4597.8    0.07       0  4699.6   0.035       0  5021.8   0.035       0
  5028.8   0.035       0
Bank Sta=5021.8,5028.8
Exp/Cntr=0.3,0.1

Type RM Length L Ch R = 1,8219,344,344,344
BEGIN DESCRIPTION:
Mapping XS edea0989
END DESCRIPTION:
XS GIS Cut Line= 3
      1635021.35      6949651.13      1635201.91      6949842.10
      1635719.59      6950852.93
#Sta/Elev= 30
  4737.9 1634.58  4746.1 1634.17  4830.0 1631.79  4900.8 1627.84  4908.1 1626.94
  4929.2 1626.41  4945.7 1622.24  4964.7 1617.78  4975.2 1617.17  4975.7 1616.67
  4982.1 1616.67  4982.6 1617.17  4999.3 1618.78  5007.3 1620.74  5015.7 1621.32
  5060.1 1622.04  5215.6 1622.05  5237.8 1621.57  5260.0 1622.19  5378.1 1622.38
  5587.4 1622.00  5647.7 1622.61  5692.7 1622.36  5715.0 1623.15  5726.4 1622.65
  5848.2 1622.98  5861.2 1623.47  5937.0 1623.30  5951.1 1623.81  6136.4 1623.58
#Mann=5,-1,0
  4737.9   0.035       0  4746.1    0.07       0  4945.7   0.035       0
  4975.2   0.035       0  4982.6   0.035       0
Bank Sta=4975.2,4982.6
Exp/Cntr=0.3,0.1

Type RM Length L Ch R = 1,7875,281,281,281
BEGIN DESCRIPTION:
Mapping XS 3bf5cc23
END DESCRIPTION:
XS GIS Cut Line= 3
      1634759.20      6949885.50      1635000.52      6950079.95
      1635274.66      6950243.05
#Sta/Elev= 30
  4689.2 1629.84  4695.7 1629.90  4766.1 1627.01  4780.5 1626.90  4801.3 1625.80
  4858.9 1624.33  4879.7 1623.10  4922.8 1621.62  4929.3 1621.17  4943.6 1618.88
  4951.6 1618.12  4966.0 1617.85  4972.4 1618.11  4979.2 1616.61  4983.1 1616.36
  4983.6 1615.86  4990.1 1615.86  4990.6 1616.36  4993.2 1616.60  4998.8 1618.07
  5002.1 1618.07  5007.6 1620.18  5029.0 1620.57  5038.8 1621.20  5050.9 1620.45
  5081.6 1620.33  5103.0 1619.84  5109.0 1619.37  5161.5 1620.81  5318.1 1621.66
#Mann=3,-1,0
  4689.2   0.035       0  4983.1   0.035       0  4990.6   0.035       0
Bank Sta=4983.1,4990.6
Exp/Cntr=0.3,0.1

Type RM Length L Ch R = 1,7594,329,329,329
BEGIN DESCRIPTION:
Mapping XS 80943923
END DESCRIPTION:
XS GIS Cut Line= 3
      1634349.33      6950013.20      1634800.86      6950262.24
      1635450.03      6950419.46
#Sta/Elev= 30
  4480.6 1625.29  4518.6 1625.53  4578.2 1624.84  4583.9 1624.24  4643.5 1623.85
  4671.0 1622.90  4687.1 1623.00  4708.9 1621.57  4746.7 1620.84  4752.4 1620.20
  4953.0 1620.15  4974.8 1619.53  4992.0 1616.44  4992.5 1615.94  4999.0 1615.94
  4999.5 1616.44  5010.8 1617.22  5044.4 1617.87  5072.5 1619.55  5093.1 1619.83
  5164.7 1619.96  5211.7 1618.70  5253.5 1619.38  5329.8 1618.58  5391.5 1620.80
  5462.6 1621.12  5467.7 1620.56  5509.6 1621.27  5556.5 1621.09  5664.2 1621.98
#Mann=3,-1,0
  4480.6   0.035       0  4992.0   0.035       0  4999.5   0.035       0
Bank Sta=4992,4999.5
Exp/Cntr=0.3,0.1

Type RM Length L Ch R = 1,7265,398,398,398
BEGIN DESCRIPTION:
Mapping XS 1526348a
END DESCRIPTION:
XS GIS Cut Line= 3
      1634283.36      6950072.22      1634908.76      6950562.18
      1635388.99      6950793.48
#Sta/Elev= 30
  4209.8 1624.07  4229.1 1623.50  4293.3 1623.28  4407.2 1620.29  4456.9 1619.57
  4599.8 1619.37  4614.2 1619.44  4620.6 1620.03  4628.7 1619.27  4643.2 1619.10
  4763.4 1619.46  4891.8 1618.96  4976.8 1618.04  4984.9 1617.54  4991.3 1617.78
  5004.3 1616.02  5018.5 1615.01  5019.0 1614.51  5025.6 1614.51  5026.1 1615.01
  5034.1 1615.40  5051.2 1617.62  5056.7 1616.98  5066.7 1616.79  5101.9 1617.28
  5119.0 1618.01  5124.6 1618.82  5141.6 1619.08  5155.5 1619.94  5537.3 1622.53
#Mann=3,-1,0
  4209.8   0.035       0  5018.5   0.035       0  5026.1   0.035       0
Bank Sta=5018.5,5026.1
Exp/Cntr=0.3,0.1

Type RM Length L Ch R = 1,6867,477,477,477
BEGIN DESCRIPTION:
Mapping XS ab8a299b
END DESCRIPTION:
XS GIS Cut Line= 3
      1634267.82      6950589.66      1634653.56      6950837.35
      1635279.98      6951012.99
#Sta/Elev= 30
  4541.1 1616.77  4545.5 1617.13  4551.4 1616.83  4660.4 1617.07  4717.9 1617.62
  4848.0 1617.30  4857.3 1617.71  4863.2 1617.22  4878.4 1617.70  4906.2 1617.05
  4941.8 1617.16  4965.6 1616.67  4987.4 1614.53  4993.4 1614.51  4993.6 1613.79
  4994.1 1613.29  5000.7 1613.29  5001.2 1613.79  5011.4 1614.34  5023.7 1614.31
  5032.2 1615.13  5115.3 1615.91  5188.0 1617.84  5271.0 1618.76  5278.0 1619.29
  5283.2 1618.88  5498.1 1621.29  5509.9 1620.94  5582.6 1621.79  5650.1 1621.76
#Mann=3,-1,0
  4541.1   0.035       0  4993.6   0.035       0  5001.2   0.035       0
Bank Sta=4993.6,5001.2
Exp/Cntr=0.3,0.1

Type RM Length L Ch R = 1,6390,370,370,370
BEGIN DESCRIPTION:
Mapping XS ee3bbb00
END DESCRIPTION:
XS GIS Cut Line= 3
      1634220.90      6950666.00      1634554.60      6951238.39
      1634790.17      6951558.12
#Sta/Elev= 30
  4341.6 1616.35  4367.1 1616.40  4376.2 1615.91  4382.0 1616.39  4419.2 1615.94
  4499.4 1615.85  4515.1 1615.41  4520.9 1615.92  4529.1 1615.46  4579.6 1615.47
  4616.9 1615.05  4638.4 1615.51  4644.9 1615.12  4740.1 1614.76  4888.0 1615.28
  4894.7 1614.86  4937.8 1614.60  4959.3 1614.07  4977.0 1611.60  4977.5 1611.10
  4984.1 1611.10  4984.6 1611.60  5001.0 1612.68  5007.0 1612.68  5017.8 1613.96
  5026.2 1614.24  5047.1 1616.32  5061.7 1616.59  5182.8 1617.25  5401.3 1617.32
#Mann=3,-1,0
  4341.6   0.035       0  4977.0   0.035       0  4984.6   0.035       0
Bank Sta=4977,4984.6
Exp/Cntr=0.3,0.1

Type RM Length L Ch R = 1,6020,341,341,341
BEGIN DESCRIPTION:
Mapping XS 1606147d
END DESCRIPTION:
XS GIS Cut Line= 3
      1634251.28      6950784.37      1634236.43      6951224.79
      1634193.29      6951468.13
#Sta/Elev= 30
  4565.0 1615.36  4648.7 1614.38  4668.7 1614.41  4698.7 1613.95  4708.7 1614.10
  4718.7 1613.76  4758.7 1613.65  4778.7 1612.11  4785.0 1611.92  4785.5 1611.42
  4792.1 1611.42  4792.6 1611.92  4828.8 1613.25  4868.8 1613.55  4901.7 1612.88
  4948.8 1613.82  4978.9 1613.25  4988.9 1612.55  4998.9 1612.28  5038.4 1612.22
  5043.5 1613.73  5049.6 1614.17  5059.7 1614.44  5110.5 1614.68  5120.6 1615.10
  5130.8 1614.92  5161.7 1615.64  5171.4 1615.42  5222.2 1615.72  5252.8 1615.36
#Mann=3,-1,0
  4565.0   0.035       0  4785.0   0.035       0  4792.6   0.035       0
Bank Sta=4785,4792.6
Exp/Cntr=0.3,0.1

Type RM Length L Ch R = 1,5679,246,246,246
BEGIN DESCRIPTION:
Mapping XS b7942bd9
END DESCRIPTION:
XS GIS Cut Line= 3
      1634204.38      6950798.32      1633906.57      6951183.13
      1633826.82      6951324.50
#Sta/Elev= 30
  4516.4 1615.09  4551.9 1614.73  4657.8 1612.42  4680.4 1612.59  4686.8 1613.00
  4693.1 1612.59  4701.3 1612.94  4786.4 1612.81  4794.2 1613.16  4807.2 1612.72
  4857.4 1612.83  4871.5 1612.30  4879.7 1612.49  4886.0 1611.89  4929.5 1611.99
  4935.8 1611.35  4958.5 1610.44  4964.8 1609.19  4975.5 1608.96  4976.0 1608.46
  4982.6 1608.46  4983.1 1608.96  4985.6 1610.25  4993.8 1611.02  5000.1 1612.76
  5015.3 1612.84  5021.1 1613.75  5052.9 1614.22  5155.5 1613.94  5165.3 1614.19
#Mann=3,-1,0
  4516.4   0.035       0  4975.5   0.035       0  4983.1   0.035       0
Bank Sta=4975.5,4983.1
Exp/Cntr=0.3,0.1

Type RM Length L Ch R = 1,5433,235,235,235
BEGIN DESCRIPTION:
Mapping XS 0328baf3
END DESCRIPTION:
XS GIS Cut Line= 3
      1634162.74      6950563.91      1633865.40      6950949.94
      1633744.32      6951221.94
#Sta/Elev= 30
  4515.2 1615.43  4581.2 1615.77  4666.3 1614.88  4672.7 1615.14  4680.9 1615.00
  4687.2 1614.46  4709.7 1614.19  4801.3 1611.23  4830.3 1611.55  4851.2 1611.24
  4901.0 1612.42  4923.7 1612.16  4944.5 1612.56  4959.0 1611.80  4973.5 1609.76
  4979.8 1609.32  5007.0 1609.06  5007.5 1608.56  5014.1 1608.56  5014.6 1609.06
  5016.3 1609.60  5022.2 1609.59  5045.0 1611.36  5068.2 1611.10  5131.7 1612.62
  5197.4 1613.16  5213.1 1613.60  5230.2 1613.29  5252.1 1613.67  5300.2 1613.56
#Mann=3,-1,0
  4515.2   0.035       0  5007.0   0.035       0  5014.6   0.035       0
Bank Sta=5007,5014.6
Exp/Cntr=0.3,0.1

Type RM Length L Ch R = 1,5198,273,273,273
BEGIN DESCRIPTION:
Mapping XS 390e3cca
END DESCRIPTION:
XS GIS Cut Line= 3
      1633627.32      6950626.08      1633690.93      6950939.53
      1633695.03      6951127.85
#Sta/Elev= 30
  4682.5 1611.92  4715.1 1611.57  4735.5 1610.93  4748.5 1610.92  4766.1 1610.44
  4799.2 1610.15  4806.9 1609.79  4837.5 1609.21  4868.1 1610.10  4900.5 1610.48
  4908.9 1610.95  4929.3 1610.51  4939.6 1609.52  4946.0 1609.28  4976.6 1608.73
  4977.1 1608.23  4983.7 1608.23  4984.2 1608.73  5000.0 1609.67  5010.8 1609.66
  5020.8 1610.00  5040.8 1609.80  5070.8 1611.10  5110.8 1611.79  5120.8 1612.27
  5130.8 1612.29  5140.8 1612.61  5170.8 1612.68  5180.8 1612.95  5190.7 1612.94
#Mann=3,-1,0
  4682.5   0.035       0  4976.6   0.035       0  4984.2   0.035       0
Bank Sta=4976.6,4984.2
Exp/Cntr=0.3,0.1

Type RM Length L Ch R = 1,4925,222,222,222
BEGIN DESCRIPTION:
Mapping XS a083b1cd
END DESCRIPTION:
XS GIS Cut Line= 3
      1633550.94      6950606.95      1633433.11      6950989.01
      1633418.99      6951290.96
#Sta/Elev= 30
  4601.2 1611.17  4638.6 1610.86  4644.2 1611.07  4671.3 1610.64  4736.6 1609.00
  4748.8 1608.43  4769.3 1608.12  4774.5 1607.61  4790.7 1608.14  4812.4 1608.18
  4839.8 1609.19  4845.1 1609.01  4853.5 1609.56  4872.5 1609.81  4937.2 1609.04
  4968.6 1608.26  4981.0 1607.52  5026.2 1607.14  5026.7 1606.64  5033.4 1606.64
  5033.9 1607.14  5040.0 1607.29  5066.4 1609.68  5071.4 1609.58  5120.1 1611.05
  5150.2 1610.98  5190.2 1611.54  5270.3 1611.53  5278.5 1611.98  5303.3 1611.44
#Mann=3,-1,0
  4601.2   0.035       0  5026.2   0.035       0  5033.9   0.035       0
Bank Sta=5026.2,5033.9
Exp/Cntr=0.3,0.1

Type RM Length L Ch R = 1,4703,308,308,308
BEGIN DESCRIPTION:
Mapping XS 1d9c07de
END DESCRIPTION:
XS GIS Cut Line= 3
      1633493.62      6950539.30      1633210.46      6950990.31
      1633219.34      6951320.56
#Sta/Elev= 30
  4470.1 1610.71  4606.5 1609.78  4648.9 1608.89  4657.5 1608.53  4670.1 1607.40
  4716.0 1606.63  4751.9 1607.22  4794.9 1608.47  4822.8 1608.59  4831.5 1609.03
  4837.4 1608.51  4858.6 1608.10  4889.2 1607.95  4904.5 1607.42  4917.3 1606.49
  4931.6 1606.08  4985.5 1605.48  4986.0 1604.98  4992.7 1604.98  4993.2 1605.48
  5020.3 1605.86  5040.3 1607.78  5060.3 1608.71  5110.4 1610.06  5160.4 1610.38
  5170.4 1610.73  5270.4 1610.73  5280.4 1611.13  5290.4 1610.79  5333.0 1610.80
#Mann=3,-1,0
  4470.1   0.035       0  4985.5   0.035       0  4993.2   0.035       0
Bank Sta=4985.5,4993.2
Exp/Cntr=0.3,0.1

Type RM Length L Ch R = 1,4395,74,74,74
BEGIN DESCRIPTION:
Mapping XS 5affe1d8
END DESCRIPTION:
XS GIS Cut Line= 3
      1632959.15      6950288.53      1632920.09      6950942.13
      1632926.60      6951237.69
#Sta/Elev= 30
  4349.4 1614.00  4378.9 1613.70  4419.0 1611.32  4459.1 1610.31  4498.5 1609.97
  4509.2 1609.50  4569.3 1609.14  4639.4 1607.91  4672.5 1607.91  4689.5 1607.56
  4709.5 1607.05  4729.5 1605.23  4769.6 1604.01  4799.7 1604.03  4836.4 1605.69
  4889.8 1606.12  4960.0 1605.64  4980.0 1604.64  5004.2 1604.20  5010.0 1603.08
  5016.2 1602.87  5016.7 1602.37  5023.4 1602.37  5023.9 1602.87  5040.0 1603.25
  5060.1 1605.76  5080.1 1606.80  5100.1 1606.83  5180.1 1608.11  5299.8 1608.84
#Mann=3,-1,0
  4349.4   0.035       0  5016.2   0.035       0  5023.9   0.035       0
Bank Sta=5016.2,5023.9
Exp/Cntr=0.3,0.1

Type RM Length L Ch R = 1,4321,471,471,471
BEGIN DESCRIPTION:
Mapping XS 03b501c3
END DESCRIPTION:
XS GIS Cut Line= 3
      1632733.89      6950427.80      1632847.18      6950942.13
      1632852.38      6951202.52
#Sta/Elev= 30
  4477.6 1610.78  4498.3 1610.96  4518.8 1609.87  4553.5 1609.03  4631.4 1608.05
  4662.1 1607.03  4682.6 1604.59  4703.1 1605.44  4733.6 1605.49  4744.0 1606.07
  4782.4 1603.92  4866.9 1603.94  4887.4 1604.95  4972.7 1605.63  4999.6 1603.09
  5010.1 1603.43  5026.3 1602.83  5026.8 1602.33  5033.5 1602.33  5034.0 1602.83
  5040.1 1602.92  5050.1 1604.36  5080.1 1605.90  5100.1 1606.01  5110.1 1604.96
  5120.1 1604.61  5145.3 1606.73  5190.2 1607.48  5250.2 1607.24  5264.7 1607.72
#Mann=3,-1,0
  4477.6   0.035       0  5026.3   0.035       0  5034.0   0.035       0
Bank Sta=5026.3,5034
Exp/Cntr=0.3,0.1

Type RM Length L Ch R = 1,3850,465,465,465
BEGIN DESCRIPTION:
Mapping XS a127799b
END DESCRIPTION:
XS GIS Cut Line= 3
      1632123.23      6950728.35      1632407.54      6951035.45
      1632728.46      6951314.23
#Sta/Elev= 30
  4584.6 1624.64  4613.7 1623.39  4649.5 1620.93  4656.3 1619.97  4663.6 1619.88
  4685.2 1616.75  4727.1 1614.07  4755.5 1610.43  4786.5 1607.80  4812.2 1605.41
  4833.2 1604.25  4840.5 1604.28  4868.9 1601.56  4875.7 1601.69  4883.0 1601.04
  4918.2 1601.34  4962.8 1600.21  4963.3 1599.71  4971.7 1599.71  4972.2 1600.21
  5010.5 1600.87  5024.7 1602.54  5052.7 1603.58  5080.7 1603.42  5116.8 1604.24
  5123.5 1603.96  5293.4 1605.01  5315.3 1605.53  5329.6 1605.15  5428.2 1606.13
#Mann=5,-1,0
  4584.6   0.035       0  4685.2    0.07       0  4786.5   0.035       0
  4962.8   0.035       0  4972.2   0.035       0
Bank Sta=4962.8,4972.2
Exp/Cntr=0.3,0.1

Type RM Length L Ch R = 1,3385,300,300,300
BEGIN DESCRIPTION:
Mapping XS f023ad69
END DESCRIPTION:
XS GIS Cut Line= 3
      1631844.81      6951226.64      1632103.90      6951298.25
      1632561.10      6951394.37
#Sta/Elev= 30
  4730.0 1619.75  4740.6 1619.61  4761.3 1618.43  4815.9 1617.09  4863.2 1615.66
  4896.2 1614.05  4902.7 1613.29  4907.9 1613.30  4916.9 1612.18  4927.3 1608.18
  4937.0 1602.73  4942.2 1602.29  4948.1 1597.75  4953.7 1597.25  4954.2 1596.75
  4962.7 1596.75  4963.2 1597.25  4976.5 1597.93  5001.9 1597.97  5018.6 1599.70
  5051.0 1601.30  5091.9 1601.83  5119.2 1601.60  5163.0 1601.90  5168.1 1601.47
  5173.6 1601.85  5224.7 1602.08  5275.8 1603.20  5362.4 1604.23  5466.0 1604.46
#Mann=5,-1,0
  4730.0   0.035       0  4815.9    0.07       0  4953.7    0.07       0
  4963.2    0.07       0  5119.2   0.035       0
Bank Sta=4953.7,4963.2
Exp/Cntr=0.3,0.1

Type RM Length L Ch R = 1,3085,316,316,316
BEGIN DESCRIPTION:
Mapping XS 93e6b292
END DESCRIPTION:
XS GIS Cut Line= 3
      1631712.94      6951506.54      1632054.11      6951582.06
      1632518.94      6951727.89
#Sta/Elev= 30
  4649.3 1618.23  4702.6 1616.75  4721.7 1615.83  4770.5 1614.70  4860.5 1611.15
  4911.6 1608.90  4938.2 1603.00  4955.2 1598.18  4979.2 1596.15  4984.6 1596.06
  4985.1 1595.56  4993.6 1595.56  4994.1 1596.06  5003.4 1596.98  5010.1 1599.05
  5020.6 1598.98  5035.8 1597.99  5041.6 1598.96  5062.5 1600.24  5103.8 1600.63
  5165.5 1601.99  5197.9 1602.29  5230.2 1602.11  5261.7 1602.63  5268.0 1602.31
  5282.6 1602.82  5300.4 1602.48  5324.6 1602.86  5356.0 1602.70  5485.9 1603.86
#Mann=5,-1,0
  4649.3   0.035       0  4860.5    0.07       0  4984.6    0.07       0
  4994.1    0.07       0  5103.8   0.035       0
Bank Sta=4984.6,4994.1
Exp/Cntr=0.3,0.1

Type RM Length L Ch R = 1,2769,306,306,306
BEGIN DESCRIPTION:
Mapping XS 20122c97
END DESCRIPTION:
XS GIS Cut Line= 3
      1631763.77      6951742.23      1632004.63      6951882.84
      1632555.42      6952043.00
#Sta/Elev= 30
  4723.0 1611.63  4746.7 1610.63  4780.3 1608.91  4817.1 1605.90  4829.1 1602.72
  4844.8 1600.35  4851.8 1599.77  4903.5 1598.52  4932.8 1597.14  4956.0 1597.36
  4962.2 1598.15  4968.0 1597.77  5001.9 1597.70  5012.7 1597.25  5018.3 1596.12
  5018.8 1595.62  5027.4 1595.62  5027.9 1596.12  5043.9 1598.71  5085.6 1600.62
  5137.7 1600.80  5158.5 1600.41  5177.8 1600.96  5183.0 1600.55  5255.3 1600.67
  5439.7 1602.70  5450.1 1602.32  5466.9 1602.84  5472.1 1602.43  5575.5 1603.34
#Mann=4,-1,0
  4723.0    0.07       0  4746.7   0.035       0  5018.3   0.035       0
  5027.9   0.035       0
Bank Sta=5018.3,5027.9
Exp/Cntr=0.3,0.1

Type RM Length L Ch R = 1,2463,364,364,364
BEGIN DESCRIPTION:
Mapping XS 5b24fb35
END DESCRIPTION:
XS GIS Cut Line= 3
      1631548.79      6952025.70      1631823.35      6952120.11
      1632331.66      6952285.58
#Sta/Elev= 30
  4710.1 1608.03  4716.7 1608.07  4727.2 1609.26  4732.5 1610.79  4737.8 1609.96
  4748.4 1607.43  4780.1 1604.24  4789.7 1602.52  4814.9 1601.01  4875.3 1599.42
  4883.4 1599.72  4888.7 1599.03  4896.4 1599.27  4945.9 1597.77  4982.4 1595.33
  5003.9 1595.08  5008.6 1594.27  5018.4 1593.93  5018.9 1593.43  5027.5 1593.43
  5028.0 1593.93  5040.5 1594.55  5054.8 1596.88  5065.3 1597.58  5104.4 1598.58
  5159.9 1598.77  5256.7 1598.21  5434.2 1600.48  5466.1 1600.28  5535.0 1601.09
#Mann=5,-1,0
  4710.1    0.07       0  4814.9   0.035       0  5018.4   0.035       0
  5028.0   0.035       0  5256.7    0.07       0
Bank Sta=5018.4,5028
Exp/Cntr=0.3,0.1

Type RM Length L Ch R = 1,2099,411,411,411
BEGIN DESCRIPTION:
Mapping XS f1998e44
END DESCRIPTION:
XS GIS Cut Line= 3
      1631380.62      6952300.66      1631637.81      6952407.00
      1632100.92      6952520.84
#Sta/Elev= 30
  4723.4 1601.85  4760.9 1600.65  4784.8 1600.43  4793.1 1599.85  4847.2 1598.30
  4856.5 1598.48  4909.7 1596.09  4922.9 1594.75  4933.6 1594.71  4939.0 1594.27
  4962.9 1594.09  4992.2 1594.49  5014.6 1593.43  5015.1 1592.93  5023.7 1592.93
  5024.2 1593.43  5040.0 1593.73  5060.6 1596.46  5155.5 1596.57  5173.9 1596.92
  5204.8 1596.69  5233.4 1597.14  5238.6 1596.56  5246.0 1596.82  5274.9 1596.25
  5307.7 1595.08  5338.6 1596.46  5348.9 1596.35  5369.5 1597.11  5478.6 1598.60
#Mann=3,-1,0
  4723.4    0.07       0  5014.6    0.07       0  5024.2    0.07       0
Bank Sta=5014.6,5024.2
Exp/Cntr=0.3,0.1

Type RM Length L Ch R = 1,1688,294,294,294
BEGIN DESCRIPTION:
Mapping XS aeba5fe8
END DESCRIPTION:
XS GIS Cut Line= 3
      1631127.92      6952541.91      1631354.53      6952652.74
      1632020.55      6952778.77
#Sta/Elev= 30
  4746.9 1600.81  4810.4 1599.50  4822.4 1598.63  4867.4 1597.79  4966.3 1594.75
  4980.0 1592.47  5005.0 1591.34  5005.5 1590.84  5014.2 1590.84  5014.7 1591.34
  5055.0 1592.34  5081.1 1592.48  5121.8 1593.78  5159.7 1594.19  5212.0 1594.15
  5217.1 1593.76  5254.1 1594.06  5294.8 1595.01  5326.8 1594.92  5335.5 1594.48
  5355.8 1595.16  5366.0 1594.37  5437.3 1593.62  5478.0 1594.38  5498.3 1595.52
  5508.5 1595.26  5528.9 1596.90  5536.2 1597.07  5640.8 1597.47  5677.0 1598.14
#Mann=3,-1,0
  4746.9    0.07       0  5005.0    0.07       0  5014.7    0.07       0
Bank Sta=5005,5014.7
Exp/Cntr=0.3,0.1

Type RM Length L Ch R = 1,1394,224,224,224
BEGIN DESCRIPTION:
Mapping XS de5a5e5f
END DESCRIPTION:
XS GIS Cut Line= 3
      1631029.97      6952612.97      1631346.81      6952945.92
      1631560.09      6953148.55
#Sta/Elev= 30
  4541.1 1599.88  4618.8 1598.42  4626.1 1597.96  4633.0 1598.16  4668.5 1596.89
  4739.3 1595.43  4746.2 1594.84  4753.5 1595.18  4817.0 1593.31  4831.1 1592.15
  4873.6 1590.56  4937.1 1590.10  4951.3 1590.59  4965.4 1590.35  4993.4 1588.94
  4993.9 1588.44  5003.5 1588.44  5004.0 1588.94  5008.1 1589.60  5014.9 1589.40
  5022.2 1590.77  5029.1 1591.49  5043.3 1592.42  5071.6 1593.29  5078.8 1594.14
  5085.7 1593.87  5107.1 1594.53  5128.2 1594.39  5199.0 1595.92  5294.9 1596.08
#Mann=3,-1,0
  4541.1    0.07       0  4993.4    0.07       0  5004.0    0.07       0
Bank Sta=4993.4,5004
Exp/Cntr=0.3,0.1
