--- Chimney Creek 1192.prj (project) ---

Proj Title=Chimney Creek 1192 Base Level Engineering
Current Plan=p01
Default Exp/Contr=0.3,0.1
English Units
Geom File=g01
Flow File=f01
Plan File=p01
BEGIN DESCRIPTION:
Chimney Creek 1192
END DESCRIPTION:

--- Chimney Creek 1192.p01 (plan) ---

Plan Title=Multiple Run
Short Identifier=Multiple
Geom File=g01
Flow File=f01
Subcritical Flow
K Sum by GR= 0
Std Step Tol= 0.01
Critical Tol= 0.01
Num of Std Step Trials= 20
Max Error Tol= 0.3
Flow Tol Ratio= 0.001
Split Flow NTrial= 30
Split Flow Tol= 0.02
Split Flow Ratio= 0.02
Log Output Level= 0
Friction Slope Method= 1
Unsteady Friction Slope Method= 2
Unsteady Bridges Friction Slope Method= 1
Parabolic Critical Depth
Global Vel Dist=  1 , 1 , 1
Global Log Level= 0
CheckData=True
Encroach Param= -1, 0, 0, 0
BEGIN DESCRIPTION:
Multiple Run
END DESCRIPTION:

--- Chimney Creek 1192.f01 (steady flow) ---

Flow Title=Multiple
Number of Profiles=7
Profile Names=10-year,25-year,50-year,1pct_min,100-year,1pct_plu,500-year
River Rch & RM= Chimney Creek 11,Reach-1,25441
     273     376     462     283     564    1125     850
River Rch & RM= Chimney Creek 11,Reach-1,23904
     311     432     532     327     652    1301     991
River Rch & RM= Chimney Creek 11,Reach-1,19346
     455     646     807     502    1002    1999    1562
River Rch & RM= Chimney Creek 11,Reach-1,17613
     572     821    1033     646    1289    2572    2033
River Rch & RM= Chimney Creek 11,Reach-1,9335
     706    1025    1302     822    1640    3271    2633
Boundary for River Rch & Prof#=Chimney Creek 11,Reach-1,1
Up Type=0
Dn Type=3
Dn Slope=0.005
Boundary for River Rch & Prof#=Chimney Creek 11,Reach-1,2
Up Type=0
Dn Type=3
Dn Slope=0.005
Boundary for River Rch & Prof#=Chimney Creek 11,Reach-1,3
Up Type=0
Dn Type=3
Dn Slope=0.005
Boundary for River Rch & Prof#=Chimney Creek 11,Reach-1,4
Up Type=0
Dn Type=3
Dn Slope=0.005
Boundary for River Rch & Prof#=Chimney Creek 11,Reach-1,5
Up Type=0
Dn Type=3
Dn Slope=0.005
Boundary for River Rch & Prof#=Chimney Creek 11,Reach-1,6
Up Type=0
Dn Type=3
Dn Slope=0.005
Boundary for River Rch & Prof#=Chimney Creek 11,Reach-1,7
Up Type=0
Dn Type=3
Dn Slope=0.005

--- Chimney Creek 1192.g01 (geometry) ---

Geom Title=Existing Conditions

River Reach=Chimney Creek 11,Reach-1
Reach XY= 30
      1701955.00      7036988.00      1701704.76      7037181.03
      1701395.02      7037048.68      1701205.07      7037256.22
      1701349.90      7037582.53      1700536.31      7038037.50
      1700239.79      7037738.24      1699756.76      7037934.70
      1699152.78      7037393.30      1698546.59      7038084.72
      1697160.47      7038643.26      1696299.12      7039886.04
      1695189.84      7039488.37      1693665.43      7039636.95
      1693153.50      7039241.46      1692913.02      7039291.31
      1692654.80      7039962.92      1692954.99      7040760.76
      1692832.12      7041611.52      1692503.50      7041934.39
      1691773.58      7042037.75      1690913.34      7041390.97
      1690475.39      7042368.15      1689663.44      7042441.40
      1689099.16      7043235.95      1687602.41      7043232.29
      1687804.79      7042569.73      1687699.53      7042143.10
      1687151.68      7042529.96      1686455.00      7041738.00

Type RM Length L Ch R = 1,25441,833,833,833
BEGIN DESCRIPTION:
Chimney Creek 1192 52.0
END DESCRIPTION:
XS GIS Cut Line= 3
      1701411.22      7036393.43      1701925.91      7037017.85
      1702369.53      7037577.44
#Sta/Elev= 30
  4190.8 1632.12  4203.9 1631.25  4224.7 1626.93  4296.4 1616.87  4395.4 1601.00
  4452.8 1594.72  4502.3 1591.06  4566.1 1587.91  4722.5 1582.19  4788.1 1580.80
  4857.6 1578.77  4871.0 1578.95  4878.9 1580.05  4893.2 1579.18  4977.9 1579.53
  4992.2 1577.72  4994.9 1576.07  4995.1 1575.57  4998.9 1576.07  5013.0 1577.25
  5021.0 1576.57  5049.9 1579.78  5070.7 1580.90  5184.4 1583.30  5198.9 1584.69
  5248.5 1584.93  5263.0 1586.23  5333.4 1587.50  5490.5 1592.29  5714.1 1600.27
#Mann=4,-1,0
  4190.8    0.07       0  4788.1   0.035       0  4994.9   0.035       0
  4998.9   0.035       0
Bank Sta=4994.9,4998.9
Exp/Cntr=0.3,0.1

Type RM Length L Ch R = 1,24608,280,280,280
BEGIN DESCRIPTION:
Mapping XS 95939f34
END DESCRIPTION:
XS GIS Cut Line= 3
      1700978.16      7036790.81      1701349.68      7037132.82
      1701959.03      7037535.58
#Sta/Elev= 30
  4495.6 1618.28  4512.7 1616.63  4519.4 1615.12  4576.2 1607.95  4611.9 1605.30
  4626.1 1602.76  4682.2 1597.09  4795.6 1588.30  4824.0 1586.46  4864.5 1585.02
  4909.1 1582.56  4937.4 1580.14  4951.6 1576.32  4965.8 1573.76  4978.0 1572.62
  4978.2 1572.12  4981.7 1572.12  4982.0 1572.62  5000.6 1573.14  5007.0 1574.94
  5022.0 1576.28  5058.1 1575.45  5094.2 1575.44  5130.3 1574.13  5181.5 1576.09
  5332.0 1576.78  5419.3 1580.06  5462.5 1583.72  5512.6 1586.88  5731.0 1592.62
#Mann=4,-1,0
  4495.6    0.07       0  4864.5   0.035       0  4978.0   0.035       0
  4982.0   0.035       0
Bank Sta=4978,4982
Exp/Cntr=0.3,0.1

Type RM Length L Ch R = 1,24328,424,424,424
BEGIN DESCRIPTION:
Mapping XS 5277d9c2
END DESCRIPTION:
XS GIS Cut Line= 3
      1700625.76      7037047.77      1701203.85      7037335.95
      1701877.47      7037549.49
#Sta/Elev= 30
  4353.4 1604.94  4406.4 1601.25  4412.0 1599.71  4428.8 1599.32  4441.9 1597.91
  4523.9 1593.40  4630.2 1589.92  4658.2 1587.48  4736.6 1585.28  4808.7 1582.90
  4837.2 1580.83  4854.0 1581.67  4859.6 1580.78  4921.2 1578.97  4949.5 1576.21
  4991.9 1572.11  4992.1 1571.61  4995.9 1572.11  5019.5 1574.26  5032.0 1574.44
  5126.8 1573.13  5218.4 1573.66  5255.9 1572.34  5344.2 1575.25  5345.9 1575.30
  5409.7 1578.20  5462.1 1582.81  5525.1 1586.44  5681.4 1590.56  5706.0 1591.18
#Mann=9,-1,0
  4353.4    0.07       0  4736.6   0.035       0  4808.7    0.07       0
  4949.5   0.035       0  4991.9   0.035       0  4995.9   0.035       0
  5344.2    0.07       0  5345.9   0.035       0  5681.4    0.07       0
Bank Sta=4991.9,4995.9
Exp/Cntr=0.3,0.1

Type RM Length L Ch R = 1,23904,372,372,372
BEGIN DESCRIPTION:
Mapping XS 3e1317ec
END DESCRIPTION:
XS GIS Cut Line= 3
      1700955.93      7037250.17      1701270.62      7037623.46
      1701497.74      7038074.46
#Sta/Elev= 30
  4512.7 1584.25  4558.9 1582.37  4566.1 1582.16  4694.6 1577.63  4708.9 1577.77
  4722.8 1576.57  4780.4 1574.11  4893.5 1573.13  4936.4 1571.46  4950.7 1570.34
  4985.9 1569.09  5004.1 1568.04  5004.4 1567.54  5008.1 1567.54  5008.4 1568.04
  5022.3 1570.94  5039.0 1571.73  5050.8 1572.77  5111.6 1574.68  5178.5 1577.64
  5207.6 1577.74  5217.5 1578.87  5223.1 1578.90  5239.8 1580.42  5245.4 1580.30
  5262.2 1581.68  5351.4 1583.26  5357.0 1582.81  5440.7 1584.15  5505.9 1584.50
#Mann=6,-1,0
  4512.7    0.07       0  4558.9   0.035       0  4566.1    0.07       0
  4722.8   0.035       0  5004.1   0.035       0  5008.4   0.035       0
Bank Sta=5004.1,5008.4
Exp/Cntr=0.3,0.1

Type RM Length L Ch R = 1,23532,347,347,347
BEGIN DESCRIPTION:
Mapping XS c593bbbc
END DESCRIPTION:
XS GIS Cut Line= 3
      1700819.23      7037283.85      1701046.01      7037886.05
      1701190.69      7038150.58
#Sta/Elev= 30
  4357.2 1584.62  4468.0 1580.58  4479.2 1579.64  4498.2 1579.49  4528.4 1578.12
  4533.8 1578.40  4543.3 1577.62  4558.7 1577.43  4613.7 1574.88  4637.2 1574.52
  4809.2 1569.18  4814.6 1569.49  4949.3 1567.95  4983.0 1565.22  4983.3 1564.72
  4987.1 1564.72  4987.3 1565.22  4992.1 1565.50  4999.1 1568.85  5004.6 1568.85
  5008.8 1571.59  5014.5 1572.36  5037.1 1574.57  5052.4 1574.56  5074.3 1577.37
  5090.4 1578.47  5112.2 1579.58  5199.5 1581.55  5215.6 1581.22  5302.2 1582.87
#Mann=4,-1,0
  4357.2    0.07       0  4637.2   0.035       0  4983.0   0.035       0
  4987.3   0.035       0
Bank Sta=4983,4987.3
Exp/Cntr=0.3,0.1

Type RM Length L Ch R = 1,23185,368,368,368
BEGIN DESCRIPTION:
Mapping XS 9bf2a96c
END DESCRIPTION:
XS GIS Cut Line= 3
      1700634.66      7037386.38      1700753.15      7037938.46
      1700880.39      7038338.35
#Sta/Elev= 30
  4439.5 1581.44  4533.2 1577.55  4543.4 1577.29  4553.7 1577.84  4574.1 1576.44
  4664.8 1573.74  4819.6 1569.29  4962.8 1567.88  4983.2 1567.14  4993.9 1565.78
  5001.4 1563.73  5026.1 1563.49  5026.4 1562.99  5030.2 1562.99  5030.5 1563.49
  5035.2 1563.57  5055.3 1568.90  5066.6 1570.48  5092.8 1572.08  5098.1 1573.15
  5125.0 1575.91  5194.7 1576.73  5221.7 1575.59  5227.0 1576.30  5234.5 1574.75
  5253.9 1573.20  5276.5 1574.33  5297.5 1576.49  5323.7 1576.91  5423.8 1580.57
#Mann=4,-1,0
  4439.5    0.07       0  4664.8   0.035       0  5026.1   0.035       0
  5030.5   0.035       0
Bank Sta=5026.1,5030.5
Exp/Cntr=0.3,0.1

Type RM Length L Ch R = 1,22817,450,450,450
BEGIN DESCRIPTION:
Mapping XS 1f0b8d2e
END DESCRIPTION:
XS GIS Cut Line= 3
      1700488.83      7037373.35      1700431.53      7038042.62
      1700439.34      7038343.20
#Sta/Elev= 30
  4332.6 1581.16  4387.4 1579.39  4434.3 1577.00  4457.7 1576.51  4598.2 1571.42
  4628.3 1570.90  4661.6 1569.65  4698.6 1567.67  4758.8 1565.50  4785.9 1565.37
  4790.9 1565.01  4809.0 1565.29  4869.2 1564.99  4939.5 1565.68  4969.6 1564.70
  4989.6 1563.62  4997.2 1562.51  4997.6 1562.01  5001.4 1562.01  5001.7 1562.51
  5009.7 1563.23  5019.7 1566.65  5029.7 1567.40  5049.7 1567.81  5059.7 1568.55
  5069.7 1569.53  5089.7 1572.46  5099.7 1573.52  5295.4 1579.90  5305.0 1580.63
#Mann=5,-1,0
  4332.6    0.07       0  4661.6   0.035       0  4997.2   0.035       0
  5001.7   0.035       0  5295.4    0.07       0
Bank Sta=4997.2,5001.7
Exp/Cntr=0.3,0.1

Type RM Length L Ch R = 1,22367,520,520,520
BEGIN DESCRIPTION:
Mapping XS 4406166d
END DESCRIPTION:
XS GIS Cut Line= 3
      1700298.07      7037389.41      1700211.27      7037739.89
      1699933.82      7038253.59
#Sta/Elev= 30
  4641.7 1578.64  4702.1 1575.78  4774.3 1573.46  4877.2 1569.47  4945.7 1566.00
  4959.6 1565.54  4990.5 1563.02  4999.2 1560.10  5003.6 1559.83  5003.9 1559.33
  5007.8 1559.33  5008.1 1559.83  5027.8 1560.79  5044.0 1562.91  5071.5 1562.17
  5093.4 1562.51  5109.6 1563.49  5137.2 1562.89  5147.7 1563.16  5153.4 1564.00
  5169.6 1562.10  5197.2 1562.18  5344.7 1565.06  5375.7 1564.97  5410.4 1569.11
  5420.9 1569.26  5442.8 1571.21  5448.4 1570.90  5464.6 1572.36  5586.6 1575.43
#Mann=5,-1,0
  4641.7   0.035       0  4774.3    0.07       0  4945.7   0.035       0
  5003.6   0.035       0  5008.1   0.035       0
Bank Sta=5003.6,5008.1
Exp/Cntr=0.3,0.1

Type RM Length L Ch R = 1,21847,296,296,296
BEGIN DESCRIPTION:
Mapping XS c15d7b85
END DESCRIPTION:
XS GIS Cut Line= 3
      1699852.17      7037246.02      1699791.41      7037939.59
      1699787.07      7038069.79
#Sta/Elev= 30
  4305.5 1576.04  4317.5 1575.50  4337.6 1573.88  4387.8 1571.36  4421.7 1570.35
  4518.3 1566.94  4578.5 1565.37  4638.8 1564.52  4715.3 1562.46  4729.1 1562.18
  4739.1 1562.42  4769.3 1561.56  4779.3 1561.76  4809.4 1561.11  4889.0 1560.89
  4929.9 1559.91  4970.0 1559.56  5017.9 1557.19  5018.2 1556.69  5022.1 1556.69
  5022.4 1557.19  5030.2 1557.30  5039.6 1558.95  5044.6 1559.36  5050.2 1561.83
  5060.2 1563.75  5080.2 1565.59  5110.2 1567.17  5128.6 1568.76  5132.0 1568.76
#Mann=6,-1,0
  4305.5    0.07       0  4421.7   0.035       0  4715.3    0.07       0
  4889.0   0.035       0  5017.9   0.035       0  5022.4   0.035       0
Bank Sta=5017.9,5022.4
Exp/Cntr=0.3,0.1

Type RM Length L Ch R = 1,21551,253,253,253
BEGIN DESCRIPTION:
Mapping XS 9c9b299a
END DESCRIPTION:
XS GIS Cut Line= 3
      1699734.03      7037425.93      1699582.97      7037768.85
      1699449.64      7038006.94
#Sta/Elev= 30
  4627.7 1566.28  4655.0 1565.40  4743.2 1562.49  4782.0 1561.77  4892.2 1558.12
  4909.6 1558.05  4925.0 1557.05  4932.9 1557.09  4938.4 1556.08  4946.9 1556.71
  4953.6 1556.31  4979.6 1555.28  4985.0 1554.32  4996.9 1554.29  4997.2 1553.79
  5001.2 1553.79  5001.5 1554.29  5007.8 1554.56  5023.8 1557.55  5035.8 1560.68
  5051.2 1562.37  5061.8 1562.72  5081.7 1563.69  5088.9 1564.82  5110.6 1565.66
  5139.0 1566.48  5172.3 1566.22  5213.3 1565.95  5245.3 1566.57  5275.3 1566.97
#Mann=9,-1,0
  4627.7   0.035       0  4655.0    0.07       0  4743.2   0.035       0
  4953.6    0.07       0  4996.9    0.07       0  5001.5    0.07       0
  5061.8   0.035       0  5172.3    0.07       0  5245.3   0.035       0
Bank Sta=4996.9,5001.5
Exp/Cntr=0.3,0.1

Type RM Length L Ch R = 1,21298,328,328,328
BEGIN DESCRIPTION:
Mapping XS f8f46025
END DESCRIPTION:
XS GIS Cut Line= 3
      1699451.03      7037234.10      1699404.15      7037590.90
      1699397.21      7037949.37
#Sta/Elev= 30
  4643.5 1570.52  4651.9 1570.94  4657.5 1569.46  4667.6 1568.23  4677.7 1567.64
  4725.6 1562.11  4748.3 1560.12  4798.7 1558.77  4809.4 1557.60  4839.1 1556.84
  4849.1 1556.19  4874.6 1555.89  4909.7 1555.85  4919.8 1555.12  4929.8 1553.85
  4959.5 1553.80  4959.8 1553.30  4963.8 1553.30  4964.1 1553.80  4970.2 1554.19
  5003.4 1554.52  5030.5 1556.00  5060.5 1557.15  5070.5 1557.17  5150.5 1559.53
  5169.6 1560.54  5216.6 1561.89  5289.3 1562.77  5350.5 1564.03  5361.9 1564.61
#Mann=6,-1,0
  4643.5    0.07       0  4874.6   0.035       0  4959.5   0.035       0
  4964.1   0.035       0  5169.6    0.07       0  5289.3   0.035       0
Bank Sta=4959.5,4964.1
Exp/Cntr=0.3,0.1

Type RM Length L Ch R = 1,20970,187,187,187
BEGIN DESCRIPTION:
Mapping XS 616f3744
END DESCRIPTION:
XS GIS Cut Line= 3
      1699074.49      7037199.36      1699158.71      7037392.11
      1699341.00      7037826.14
#Sta/Elev= 30
  4791.1 1582.35  4822.4 1579.00  4881.1 1574.67  4920.6 1570.46  4933.3 1568.38
  4942.4 1565.00  4956.7 1562.33  4974.7 1556.31  4980.1 1556.15  4986.0 1553.26
  4998.8 1548.43  5001.2 1547.20  5001.6 1546.70  5005.6 1546.70  5005.9 1547.20
  5018.7 1549.68  5032.8 1550.50  5051.1 1553.51  5062.1 1554.33  5141.9 1555.45
  5243.6 1556.27  5300.7 1556.81  5310.4 1558.02  5315.8 1557.29  5322.4 1558.45
  5345.0 1560.20  5368.8 1557.81  5392.5 1558.97  5447.6 1559.98  5472.2 1561.19
#Mann=7,-1,0
  4791.1    0.07       0  4998.8   0.035       0  5001.2   0.035       0
  5005.9   0.035       0  5141.9    0.07       0  5243.6   0.035       0
  5447.6    0.07       0
Bank Sta=5001.2,5005.9
Exp/Cntr=0.3,0.1

Type RM Length L Ch R = 1,20783,165,165,165
BEGIN DESCRIPTION:
Mapping XS fe1255fa
END DESCRIPTION:
XS GIS Cut Line= 3
      1698925.97      7037362.84      1699034.32      7037510.08
      1699237.07      7037806.57
#Sta/Elev= 30
  4818.1 1573.20  4821.6 1572.01  4836.2 1570.85  4842.5 1570.71  4878.0 1565.82
  4907.2 1562.93  4913.4 1562.74  4921.9 1560.96  4928.1 1558.96  4936.2 1557.26
  4942.7 1555.48  4963.6 1551.48  4972.0 1549.24  4985.9 1549.00  4992.9 1548.16
  5000.9 1547.86  5005.4 1546.42  5005.7 1545.92  5009.7 1545.92  5010.1 1546.42
  5022.6 1548.85  5030.0 1550.68  5034.7 1551.90  5043.6 1552.75  5049.7 1553.29
  5064.6 1553.87  5172.2 1554.62  5180.1 1555.11  5265.0 1556.30  5360.1 1558.93
#Mann=4,-1,0
  4818.1    0.07       0  5005.4    0.07       0  5010.1    0.07       0
  5030.0   0.035       0
Bank Sta=5005.4,5010.1
Exp/Cntr=0.3,0.1

Type RM Length L Ch R = 1,20618,155,155,155
BEGIN DESCRIPTION:
Mapping XS fe519627
END DESCRIPTION:
XS GIS Cut Line= 3
      1698819.27      7037516.69      1698917.22      7037625.06
      1699117.23      7037868.83
#Sta/Elev= 30
  4853.4 1562.77  4872.4 1562.17  4886.6 1561.05  4950.1 1548.01  4957.6 1546.68
  4969.4 1546.01  4969.7 1545.51  4973.8 1545.51  4974.2 1546.01  4978.5 1546.63
  4992.7 1546.43  4998.1 1549.15  5011.5 1550.10  5070.7 1550.74  5092.9 1551.51
  5099.4 1551.08  5106.8 1552.14  5113.7 1552.46  5148.9 1553.23  5156.8 1552.32
  5163.2 1552.69  5171.1 1552.21  5177.6 1552.55  5184.4 1554.14  5220.6 1555.40
  5227.1 1555.19  5235.0 1555.77  5255.8 1556.19  5284.5 1557.43  5314.8 1558.00
#Mann=4,-1,0
  4853.4    0.07       0  4969.4    0.07       0  4974.2    0.07       0
  5011.5   0.035       0
Bank Sta=4969.4,4974.2
Exp/Cntr=0.3,0.1

Type RM Length L Ch R = 1,20463,152,152,152
BEGIN DESCRIPTION:
Mapping XS d463e7ad
END DESCRIPTION:
XS GIS Cut Line= 3
      1698688.73      7037577.82      1698808.88      7037736.17
      1699008.77      7038013.10
#Sta/Elev= 30
  4802.7 1557.66  4807.0 1557.86  4850.6 1555.92  4865.2 1555.85  4889.6 1554.36
  4892.3 1554.33  4900.6 1553.01  4906.8 1553.03  4915.1 1551.45  4935.9 1549.19
  4942.2 1547.63  4956.8 1546.07  4962.6 1545.88  4963.0 1545.38  4967.1 1545.38
  4967.4 1545.88  4992.1 1547.57  5021.3 1548.02  5028.4 1547.58  5065.4 1549.38
  5107.2 1550.69  5151.4 1551.45  5157.5 1552.02  5172.2 1552.46  5178.4 1553.13
  5207.8 1553.89  5264.3 1556.63  5279.0 1556.85  5293.7 1557.84  5343.0 1559.50
#Mann=4,-1,0
  4802.7    0.07       0  4889.6   0.035       0  4962.6   0.035       0
  4967.4   0.035       0
Bank Sta=4962.6,4967.4
Exp/Cntr=0.3,0.1

Type RM Length L Ch R = 1,20311,112,112,112
BEGIN DESCRIPTION:
Mapping XS b07ca32b
END DESCRIPTION:
XS GIS Cut Line= 3
      1698630.52      7037728.44      1698700.83      7037843.03
      1698826.33      7038059.66
#Sta/Elev= 30
  4866.2 1550.86  4876.5 1550.65  4905.1 1549.91  4912.6 1549.07  4926.4 1548.53
  4963.1 1547.91  4984.4 1545.14  4991.6 1545.09  4991.9 1544.59  4996.0 1544.59
  4996.4 1545.09  4999.8 1545.85  5021.3 1546.65  5042.9 1546.78  5064.4 1545.80
  5074.4 1545.98  5080.1 1547.59  5087.3 1548.04  5095.9 1547.75  5101.7 1548.52
  5123.2 1549.69  5132.0 1549.31  5139.0 1549.23  5145.1 1548.16  5182.0 1549.01
  5191.3 1549.64  5197.8 1550.94  5203.6 1550.16  5226.0 1552.55  5251.0 1554.04
#Mann=5,-1,0
  4866.2    0.07       0  4876.5   0.035       0  4991.6   0.035       0
  4996.4   0.035       0  5132.0    0.07       0
Bank Sta=4991.6,4996.4
Exp/Cntr=0.3,0.1

Type RM Length L Ch R = 1,20199,241,241,241
BEGIN DESCRIPTION:
Mapping XS 3162e407
END DESCRIPTION:
XS GIS Cut Line= 3
      1698544.03      7037835.70      1698621.14      7037922.19
      1698722.71      7038108.66
#Sta/Elev= 30
  4884.5 1547.46  4893.9 1547.72  4908.1 1547.46  4914.8 1547.66  4922.3 1547.56
  4943.2 1548.07  4964.9 1547.85  4979.1 1547.29  4985.8 1547.37  4993.4 1547.10
  4999.5 1545.52  5007.0 1544.84  5037.6 1545.02  5043.3 1545.26  5052.5 1545.07
  5065.2 1544.20  5072.9 1544.08  5073.3 1543.58  5077.4 1543.58  5077.7 1544.08
  5081.3 1545.08  5087.0 1546.28  5105.4 1547.65  5125.0 1548.27  5155.0 1550.00
  5168.7 1551.19  5184.8 1553.48  5200.6 1554.04  5206.6 1554.79  5212.7 1555.01
#Mann=4,-1,0
  4884.5   0.035       0  5072.9   0.035       0  5077.7   0.035       0
  5105.4    0.07       0
Bank Sta=5072.9,5077.7
Exp/Cntr=0.3,0.1

Type RM Length L Ch R = 1,19958,142,142,142
BEGIN DESCRIPTION:
Mapping XS 47f46f69
END DESCRIPTION:
XS GIS Cut Line= 3
      1698557.05      7037900.24      1698506.28      7038090.31
      1698474.47      7038254.52
#Sta/Elev= 30
  4804.7 1547.29  4864.5 1547.02  4905.1 1545.64  4910.3 1544.61  4916.2 1545.44
  4926.6 1545.84  4950.4 1545.87  4957.6 1545.67  4968.0 1544.53  4978.3 1544.32
  4985.3 1542.48  4990.4 1542.92  4997.7 1542.25  5006.9 1542.22  5007.2 1541.72
  5011.3 1541.72  5011.7 1542.22  5019.5 1544.88  5029.2 1546.34  5034.6 1546.03
  5060.2 1547.02  5080.6 1549.75  5086.3 1551.76  5091.4 1550.91  5100.9 1552.84
  5121.3 1554.32  5131.5 1555.68  5138.1 1557.16  5143.2 1556.68  5168.7 1558.99
#Mann=4,-1,0
  4804.7   0.035       0  5006.9   0.035       0  5011.7   0.035       0
  5029.2    0.07       0
Bank Sta=5006.9,5011.7
Exp/Cntr=0.3,0.1

Type RM Length L Ch R = 1,19816,112,112,112
BEGIN DESCRIPTION:
Mapping XS a3171e18
END DESCRIPTION:
XS GIS Cut Line= 3
      1698279.55      7037765.55      1698381.98      7038039.00
      1698440.08      7038268.76
#Sta/Elev= 30
  4709.4 1549.59  4744.3 1548.88  4763.9 1549.66  4769.2 1548.76  4776.1 1549.47
  4818.8 1547.38  4824.4 1545.69  4840.2 1544.00  4849.4 1543.90  4861.5 1544.79
  4885.0 1544.53  4915.2 1545.38  4934.8 1545.21  4940.2 1545.78  4970.4 1544.61
  4979.0 1543.06  4987.3 1542.67  4987.6 1542.17  4991.7 1542.17  4992.1 1542.67
  4995.4 1543.56  5030.1 1544.61  5076.3 1544.22  5082.9 1543.54  5108.4 1544.85
  5144.8 1545.50  5158.4 1547.07  5165.4 1549.47  5175.7 1552.03  5238.4 1558.75
#Mann=4,-1,0
  4709.4   0.035       0  4987.3   0.035       0  4992.1   0.035       0
  5108.4    0.07       0
Bank Sta=4987.3,4992.1
Exp/Cntr=0.3,0.1

Type RM Length L Ch R = 1,19704,138,138,138
BEGIN DESCRIPTION:
Mapping XS 6d302a29
END DESCRIPTION:
XS GIS Cut Line= 3
      1698126.76      7037842.80      1698278.69      7038065.04
      1698440.49      7038327.22
#Sta/Elev= 30
  4731.8 1550.10  4812.6 1548.26  4863.4 1546.68  4899.3 1544.79  4914.2 1544.96
  4920.3 1543.31  4929.2 1543.31  4932.8 1540.28  4933.2 1539.78  4937.3 1539.78
  4937.6 1540.28  4950.1 1540.63  4956.2 1541.28  4971.1 1541.61  4986.0 1541.30
  4992.5 1540.62  5006.9 1541.73  5016.2 1542.14  5022.3 1541.94  5028.2 1542.64
  5059.0 1543.76  5111.3 1544.70  5138.2 1544.48  5159.5 1544.83  5169.0 1545.95
  5190.3 1552.47  5226.9 1555.41  5239.5 1557.19  5298.3 1560.20  5309.1 1561.21
#Mann=4,-1,0
  4731.8   0.035       0  4932.8   0.035       0  4937.6   0.035       0
  5111.3    0.07       0
Bank Sta=4932.8,4937.6
Exp/Cntr=0.3,0.1

Type RM Length L Ch R = 1,19566,220,220,220
BEGIN DESCRIPTION:
Mapping XS fcc061c5
END DESCRIPTION:
XS GIS Cut Line= 3
      1697990.94      7037977.58      1698181.06      7038162.50
      1698381.19      7038379.88
#Sta/Elev= 30
  4735.2 1548.52  4936.3 1543.43  4952.9 1543.55  4964.6 1542.98  4971.7 1541.76
  4984.2 1540.64  4997.3 1539.68  4997.6 1539.18  5001.7 1539.18  5002.1 1539.68
  5021.5 1539.78  5035.1 1541.19  5042.5 1541.49  5049.3 1542.47  5065.6 1543.18
  5077.7 1543.30  5091.8 1542.94  5106.0 1543.64  5120.2 1545.33  5127.6 1547.30
  5134.4 1548.27  5141.8 1551.08  5148.6 1551.81  5176.9 1553.31  5219.4 1557.38
  5233.6 1557.68  5240.4 1558.26  5276.2 1559.60  5290.3 1561.03  5295.9 1562.19
#Mann=6,-1,0
  4735.2   0.035       0  4952.9    0.07       0  4984.2   0.035       0
  4997.3   0.035       0  5002.1   0.035       0  5065.6    0.07       0
Bank Sta=4997.3,5002.1
Exp/Cntr=0.3,0.1

Type RM Length L Ch R = 1,19346,298,298,298
BEGIN DESCRIPTION:
Mapping XS ea4adc9d
END DESCRIPTION:
XS GIS Cut Line= 3
      1697805.22      7038040.14      1698050.85      7038332.64
      1698307.77      7038580.01
#Sta/Elev= 30
  4619.1 1548.47  4624.7 1547.98  4631.2 1548.28  4668.4 1547.11  4844.5 1542.43
  4858.8 1541.11  4865.4 1541.40  4922.6 1540.90  4957.7 1539.48  4961.2 1538.94
  4976.4 1537.21  4976.9 1536.71  4982.6 1536.71  4983.1 1537.21  4994.1 1537.38
  5000.4 1538.18  5007.7 1540.29  5043.2 1544.31  5064.3 1548.98  5071.5 1549.53
  5113.9 1550.74  5170.5 1555.37  5219.9 1557.21  5227.1 1557.72  5241.3 1559.98
  5262.4 1561.56  5269.6 1561.91  5276.5 1561.52  5283.7 1562.29  5357.7 1564.48
#Mann=5,-1,0
  4619.1    0.07       0  4668.4   0.035       0  4961.2    0.07       0
  4976.4    0.07       0  4983.1    0.07       0
Bank Sta=4976.4,4983.1
Exp/Cntr=0.3,0.1

Type RM Length L Ch R = 1,19048,322,322,322
BEGIN DESCRIPTION:
Mapping XS ca238bf6
END DESCRIPTION:
XS GIS Cut Line= 3
      1697555.31      7038081.15      1697772.33      7038391.49
      1698067.47      7038842.87
#Sta/Elev= 30
  4625.2 1562.65  4651.3 1557.37  4681.0 1554.38  4708.0 1549.35  4760.1 1545.45
  4844.9 1541.41  4859.8 1539.25  4880.7 1538.49  4889.4 1537.33  4931.3 1538.53
  4946.1 1537.49  4967.0 1537.42  4981.9 1536.21  4984.6 1535.42  4985.1 1534.92
  4991.4 1535.42  4996.7 1535.51  5005.8 1537.27  5007.4 1537.77  5011.7 1539.13
  5017.8 1539.67  5075.1 1539.70  5161.8 1542.30  5198.7 1543.61  5226.7 1545.51
  5234.9 1545.09  5364.6 1552.64  5429.8 1555.66  5479.2 1559.86  5543.2 1561.41
#Mann=7,-1,0
  4625.2    0.07       0  4760.1   0.035       0  4984.6   0.035       0
  4991.4   0.035       0  5005.8    0.07       0  5007.4   0.035       0
  5161.8    0.07       0
Bank Sta=4984.6,4991.4
Exp/Cntr=0.3,0.1

Type RM Length L Ch R = 1,18726,364,364,364
BEGIN DESCRIPTION:
Mapping XS ad5bd5a4
END DESCRIPTION:
XS GIS Cut Line= 3
      1697274.32      7038258.05      1697537.96      7038457.68
      1697978.48      7038859.14
#Sta/Elev= 30
  4671.4 1574.92  4674.9 1574.92  4700.4 1570.60  4729.0 1567.99  4743.6 1564.65
  4772.6 1560.67  4799.3 1555.11  4835.3 1547.68  4864.2 1540.44  4877.6 1539.38
  4943.3 1538.04  4989.8 1534.57  4990.3 1534.07  4996.1 1534.07  4996.6 1534.57
  5007.4 1535.39  5035.8 1535.90  5070.9 1538.75  5085.1 1539.23  5219.6 1539.81
  5288.2 1541.30  5347.3 1544.74  5404.0 1546.81  5425.0 1549.48  5453.4 1551.99
  5495.9 1553.19  5524.3 1555.53  5545.2 1556.28  5573.6 1558.27  5598.1 1558.90
#Mann=7,-1,0
  4671.4    0.07       0  4700.4   0.035       0  4799.3    0.07       0
  4877.6   0.035       0  4989.8   0.035       0  4996.6   0.035       0
  5288.2    0.07       0
Bank Sta=4989.8,4996.6
Exp/Cntr=0.3,0.1

Type RM Length L Ch R = 1,18362,301,301,301
BEGIN DESCRIPTION:
Mapping XS 3f98f272
END DESCRIPTION:
XS GIS Cut Line= 3
      1697012.49      7038452.87      1697255.57      7038634.09
      1697874.04      7038935.73
#Sta/Elev= 30
  4697.9 1576.55  4717.3 1573.22  4761.1 1569.15  4767.3 1567.70  4796.5 1564.85
  4802.8 1563.31  4846.6 1557.88  4867.4 1553.85  4882.0 1552.31  4888.3 1550.12
  4896.6 1548.85  4925.5 1545.77  4932.1 1544.34  4938.3 1541.47  4946.7 1537.07
  4952.9 1532.45  4957.9 1529.95  4958.4 1529.45  4964.7 1529.95  4988.3 1533.68
  5003.3 1535.18  5041.8 1536.54  5100.6 1536.51  5234.1 1538.35  5250.2 1537.63
  5370.5 1540.10  5413.5 1540.93  5534.5 1545.34  5588.1 1549.41  5689.2 1553.62
#Mann=5,-1,0
  4697.9    0.07       0  4957.9    0.07       0  4964.7    0.07       0
  5003.3   0.035       0  5370.5    0.07       0
Bank Sta=4957.9,4964.7
Exp/Cntr=0.3,0.1

Type RM Length L Ch R = 1,18061,448,448,448
BEGIN DESCRIPTION:
Mapping XS 6b562b7d
END DESCRIPTION:
XS GIS Cut Line= 3
      1696746.66      7038614.98      1697042.26      7038803.80
      1697919.87      7039003.02
#Sta/Elev= 30
  4651.5 1568.00  4660.9 1567.76  4666.9 1566.48  4682.1 1566.92  4688.0 1565.74
  4703.2 1565.93  4724.4 1563.83  4791.2 1560.44  4848.7 1555.50  4875.8 1552.14
  4898.7 1550.82  4927.4 1546.00  4957.9 1543.76  4969.9 1539.59  4979.0 1537.86
  4998.8 1530.31  4999.3 1529.81  5005.7 1530.31  5048.0 1532.92  5090.6 1535.01
  5199.9 1534.63  5240.9 1535.79  5268.1 1535.12  5292.2 1537.33  5394.7 1537.94
  5612.7 1541.43  5743.4 1548.49  5859.1 1553.33  5876.7 1555.75  5902.2 1557.07
#Mann=5,-1,0
  4651.5    0.07       0  4998.8    0.07       0  5005.7    0.07       0
  5048.0   0.035       0  5612.7    0.07       0
Bank Sta=4998.8,5005.7
Exp/Cntr=0.3,0.1

Type RM Length L Ch R = 1,17613,284,284,284
BEGIN DESCRIPTION:
Mapping XS 23921673
END DESCRIPTION:
XS GIS Cut Line= 3
      1696727.96      7038849.65      1696949.30      7039183.83
      1697347.71      7039452.91
#Sta/Elev= 30
  4599.8 1553.10  4681.9 1549.31  4690.9 1548.27  4712.0 1544.26  4748.1 1541.46
  4754.1 1540.41  4769.1 1536.08  4777.7 1534.25  4790.2 1532.73  4813.7 1531.47
  4841.3 1532.08  4869.4 1531.85  4928.6 1529.83  4950.9 1530.00  4957.7 1529.37
  4967.1 1527.35  4967.6 1526.85  4973.8 1526.85  4974.3 1527.35  4979.7 1527.74
  4987.4 1529.34  5000.1 1531.84  5021.3 1533.00  5167.6 1535.74  5216.1 1537.26
  5303.0 1541.47  5324.0 1541.82  5360.0 1543.83  5389.9 1547.45  5481.4 1551.15
#Mann=7,-1,0
  4599.8    0.07       0  4869.4   0.035       0  4950.9    0.07       0
  4967.1   0.035       0  4974.3    0.07       0  4987.4   0.035       0
  5167.6    0.07       0
Bank Sta=4967.1,4974.3
Exp/Cntr=0.3,0.1

Type RM Length L Ch R = 1,17329,735,735,735
BEGIN DESCRIPTION:
Mapping XS 949b0dc5
END DESCRIPTION:
XS GIS Cut Line= 3
      1696521.97      7038670.16      1696667.37      7039195.35
      1697283.08      7040183.95
#Sta/Elev= 30
  4460.6 1562.41  4561.9 1557.30  4756.3 1549.10  4821.5 1547.14  4873.4 1541.99
  4935.5 1539.61  4966.3 1534.89  4974.9 1531.76  4980.1 1528.12  5000.7 1523.76
  5001.2 1523.26  5007.9 1523.76  5033.8 1529.02  5055.8 1530.07  5164.8 1529.13
  5201.4 1530.76  5274.5 1529.86  5350.3 1531.33  5463.4 1534.13  5491.7 1537.02
  5579.0 1541.55  5703.7 1553.28  5877.6 1560.72  5941.3 1566.18  6029.8 1570.19
  6066.4 1575.51  6072.3 1578.06  6103.0 1580.55  6108.9 1582.42  6170.2 1586.76
#Mann=7,-1,0
  4460.6    0.07       0  4561.9   0.035       0  4756.3    0.07       0
  4966.3   0.035       0  5000.7   0.035       0  5007.9   0.035       0
  5350.3    0.07       0
Bank Sta=5000.7,5007.9
Exp/Cntr=0.3,0.1

Type RM Length L Ch R = 1,16594,397,397,397
BEGIN DESCRIPTION:
Mapping XS 2a66a611
END DESCRIPTION:
XS GIS Cut Line= 3
      1696276.37      7038954.84      1696373.59      7039824.64
      1696467.25      7040353.60
#Sta/Elev= 30
  4128.8 1547.29  4298.0 1542.09  4360.2 1539.94  4568.9 1533.47  4735.7 1527.70
  4836.3 1526.00  4856.5 1524.57  4926.9 1525.20  4947.0 1524.42  4971.9 1522.07
  5013.8 1521.35  5032.9 1520.30  5033.4 1519.80  5040.6 1520.30  5041.9 1521.68
  5048.0 1522.81  5095.9 1526.21  5139.4 1534.26  5155.1 1535.68  5214.2 1538.32
  5261.3 1542.43  5291.8 1543.15  5322.2 1545.87  5327.4 1547.06  5352.7 1548.50
  5386.6 1548.73  5440.7 1551.34  5499.8 1552.19  5533.3 1553.76  5541.2 1554.28
#Mann=8,-1,0
  4128.8    0.07       0  4298.0   0.035       0  4360.2    0.07       0
  4568.9   0.035       0  5013.8    0.07       0  5032.9   0.035       0
  5040.6    0.07       0  5533.3   0.035       0
Bank Sta=5032.9,5040.6
Exp/Cntr=0.3,0.1

Type RM Length L Ch R = 1,16197,485,485,485
BEGIN DESCRIPTION:
Mapping XS da45df35
END DESCRIPTION:
XS GIS Cut Line= 3
      1695995.12      7039065.99      1696017.69      7039840.26
      1696040.26      7040421.83
#Sta/Elev= 30
  4227.7 1551.97  4295.4 1549.75  4349.8 1546.97  4379.8 1544.72  4409.8 1541.18
  4469.8 1538.58  4522.0 1533.71  4709.9 1526.79  4920.0 1522.86  4970.0 1522.84
  4980.0 1522.08  4990.0 1518.59  5000.4 1517.19  5010.0 1517.83  5026.2 1516.49
  5026.7 1515.99  5033.9 1516.49  5050.1 1518.22  5058.5 1520.23  5063.5 1519.37
  5080.1 1525.77  5090.1 1530.94  5110.1 1537.36  5150.1 1543.83  5180.2 1547.10
  5240.2 1549.07  5320.9 1553.20  5338.8 1553.81  5426.3 1556.56  5584.3 1564.09
#Mann=9,-1,0
  4227.7   0.035       0  4295.4    0.07       0  4522.0   0.035       0
  5000.4    0.07       0  5026.2   0.035       0  5033.9    0.07       0
  5320.9   0.035       0  5338.8    0.07       0  5426.3   0.035       0
Bank Sta=5026.2,5033.9
Exp/Cntr=0.3,0.1

Type RM Length L Ch R = 1,15712,360,360,360
BEGIN DESCRIPTION:
Mapping XS a94f7401
END DESCRIPTION:
XS GIS Cut Line= 3
      1695833.65      7039062.51      1695561.09      7039751.72
      1695540.26      7040302.08
#Sta/Elev= 30
  4263.1 1549.77  4382.8 1547.02  4419.6 1545.51  4473.3 1539.77  4537.8 1537.84
  4549.5 1536.98  4580.9 1532.65  4621.7 1530.37  4627.9 1530.19  4652.2 1526.78
  4676.6 1525.36  4795.9 1522.03  4838.8 1521.60  4873.9 1520.05  4882.0 1520.78
  4914.2 1518.90  4922.6 1517.10  4932.5 1516.80  4968.0 1516.18  5009.7 1516.73
  5016.6 1515.17  5017.1 1514.67  5024.4 1515.17  5029.3 1518.34  5070.6 1521.76
  5100.0 1527.00  5350.8 1537.97  5390.8 1540.41  5450.8 1546.12  5555.0 1552.11
#Mann=8,-1,0
  4263.1   0.035       0  4382.8    0.07       0  4621.7   0.035       0
  4932.5    0.07       0  5009.7   0.035       0  5016.6    0.07       0
  5024.4   0.035       0  5100.0    0.07       0
Bank Sta=5016.6,5024.4
Exp/Cntr=0.3,0.1

Type RM Length L Ch R = 1,15352,341,341,341
BEGIN DESCRIPTION:
Mapping XS cd258952
END DESCRIPTION:
XS GIS Cut Line= 3
      1695264.22      7039003.45      1695272.90      7039564.22
      1695309.36      7040250.02
#Sta/Elev= 30
  4447.7 1549.02  4522.0 1543.56  4550.7 1541.02  4562.3 1539.17  4582.3 1537.60
  4642.3 1534.27  4672.3 1531.50  4732.3 1528.64  4802.3 1521.28  4825.3 1520.32
  4882.3 1518.28  4892.3 1515.96  4902.3 1514.82  5002.3 1514.19  5018.4 1513.29
  5018.9 1512.79  5026.3 1513.29  5044.4 1513.53  5074.6 1514.10  5112.5 1516.26
  5122.5 1515.68  5132.5 1516.43  5139.9 1517.93  5282.7 1523.59  5314.1 1525.47
  5402.9 1528.74  5513.0 1535.11  5593.1 1540.72  5623.2 1544.35  5695.3 1549.84
#Mann=9,-1,0
  4447.7    0.07       0  4522.0   0.035       0  4550.7    0.07       0
  4825.3   0.035       0  5018.4   0.035       0  5026.3   0.035       0
  5044.4    0.07       0  5074.6   0.035       0  5314.1    0.07       0
Bank Sta=5018.4,5026.3
Exp/Cntr=0.3,0.1

Type RM Length L Ch R = 1,15011,748,748,748
BEGIN DESCRIPTION:
Mapping XS d47663c8
END DESCRIPTION:
XS GIS Cut Line= 3
      1694949.08      7039027.40      1694975.13      7039544.77
      1695015.06      7040211.45
#Sta/Elev= 30
  4488.5 1558.54  4529.2 1554.92  4619.3 1550.97  4629.3 1549.27  4669.3 1546.23
  4729.4 1540.01  4759.4 1538.43  4769.5 1537.34  4789.5 1533.28  4819.5 1530.75
  4839.5 1527.39  4889.6 1514.76  4899.6 1513.07  4904.6 1513.43  4929.7 1510.95
  4975.6 1509.26  4976.1 1508.76  4983.8 1509.26  4989.7 1509.56  5005.6 1513.27
  5072.8 1515.67  5200.1 1519.08  5220.1 1518.52  5270.2 1520.98  5355.8 1526.87
  5390.4 1529.30  5470.6 1532.49  5587.8 1540.79  5610.8 1541.52  5674.4 1547.24
#Mann=5,-1,0
  4488.5    0.07       0  4975.6    0.07       0  4983.8    0.07       0
  5072.8   0.035       0  5355.8    0.07       0
Bank Sta=4975.6,4983.8
Exp/Cntr=0.3,0.1

Type RM Length L Ch R = 1,14263,289,289,289
BEGIN DESCRIPTION:
Mapping XS 5adbbde0
END DESCRIPTION:
XS GIS Cut Line= 3
      1694429.56      7038959.68      1694316.71      7039597.73
      1694334.07      7040359.48
#Sta/Elev= 30
  4362.1 1552.36  4401.0 1551.19  4416.6 1549.18  4461.9 1546.64  4512.7 1540.53
  4563.5 1537.92  4589.1 1534.21  4695.5 1528.89  4726.0 1525.25  4827.5 1518.76
  4868.2 1517.60  4879.8 1516.45  4918.9 1508.45  4959.5 1507.68  4990.8 1503.91
  4996.0 1503.35  4996.5 1502.85  5004.3 1503.35  5007.6 1504.59  5080.3 1509.92
  5155.0 1510.28  5300.4 1513.48  5340.4 1519.71  5390.4 1525.07  5440.4 1532.28
  5470.4 1534.26  5490.4 1538.62  5520.5 1541.87  5540.5 1545.69  5772.0 1558.13
#Mann=4,-1,0
  4362.1    0.07       0  4990.8   0.035       0  4996.0   0.035       0
  5004.3   0.035       0
Bank Sta=4996,5004.3
Exp/Cntr=0.3,0.1

Type RM Length L Ch R = 1,13974,271,271,271
BEGIN DESCRIPTION:
Mapping XS b3ceacfe
END DESCRIPTION:
XS GIS Cut Line= 3
      1694308.44      7038870.33      1694027.21      7039592.52
      1694037.63      7040273.03
#Sta/Elev= 30
  4230.0 1551.25  4278.3 1549.72  4377.7 1544.42  4417.0 1539.86  4463.6 1537.08
  4485.1 1532.44  4538.7 1529.35  4592.4 1523.70  4646.0 1519.72  4718.8 1515.82
  4742.6 1515.79  4754.0 1514.20  4866.0 1510.11  4947.0 1508.19  4957.2 1507.30
  4966.2 1503.91  4971.5 1505.27  4974.5 1503.22  4975.0 1502.72  4982.8 1503.22
  5030.5 1503.79  5040.5 1505.83  5150.5 1506.97  5240.5 1511.13  5510.6 1532.98
  5520.6 1534.38  5540.6 1539.19  5580.6 1543.23  5620.6 1545.56  5685.6 1546.93
#Mann=4,-1,0
  4230.0    0.07       0  4866.0   0.035       0  4974.5   0.035       0
  4982.8   0.035       0
Bank Sta=4974.5,4982.8
Exp/Cntr=0.3,0.1

Type RM Length L Ch R = 1,13703,373,373,373
BEGIN DESCRIPTION:
Mapping XS 52e7c9fb
END DESCRIPTION:
XS GIS Cut Line= 3
      1693650.48      7038688.03      1693775.47      7039644.60
      1693952.15      7040254.32
#Sta/Elev= 30
  4041.9 1538.02  4116.4 1535.25  4142.7 1530.07  4223.4 1524.31  4302.6 1516.40
  4348.2 1514.28  4384.8 1508.66  4418.9 1509.22  4463.7 1508.76  4546.1 1508.06
  4653.8 1504.72  4959.5 1506.46  4999.9 1502.63  5024.3 1503.44  5047.6 1501.29
  5048.1 1500.79  5055.9 1501.29  5083.0 1501.89  5091.5 1504.85  5096.7 1503.54
  5103.8 1507.30  5130.3 1514.21  5135.5 1513.01  5197.4 1519.24  5202.6 1518.49
  5308.6 1531.06  5437.0 1532.92  5458.5 1534.57  5492.1 1540.20  5641.4 1543.85
#Mann=6,-1,0
  4041.9    0.07       0  4302.6   0.035       0  4418.9    0.07       0
  4463.7   0.035       0  5047.6   0.035       0  5055.9   0.035       0
Bank Sta=5047.6,5055.9
Exp/Cntr=0.3,0.1

Type RM Length L Ch R = 1,13330,666,666,666
BEGIN DESCRIPTION:
Mapping XS 8ca2e478
END DESCRIPTION:
XS GIS Cut Line= 3
      1693218.19      7038771.35      1693461.24      7039493.56
      1693742.47      7039970.97
#Sta/Elev= 30
  4243.9 1541.60  4252.9 1539.41  4279.1 1540.39  4284.4 1538.48  4373.6 1535.72
  4378.9 1533.45  4410.4 1530.17  4468.1 1527.30  4567.9 1513.31  4594.1 1507.65
  4638.2 1505.11  4746.4 1499.12  4751.7 1500.85  4773.7 1498.01  4774.2 1497.51
  4782.0 1498.01  4877.7 1498.66  4926.2 1501.69  5011.4 1499.12  5020.0 1501.02
  5025.8 1499.77  5041.5 1505.55  5047.3 1503.71  5062.9 1504.10  5078.6 1507.82
  5143.0 1509.80  5158.6 1513.79  5195.7 1517.71  5334.3 1524.89  5560.0 1531.71
#Mann=4,-1,0
  4243.9    0.07       0  4638.2   0.035       0  4773.7   0.035       0
  4782.0   0.035       0
Bank Sta=4773.7,4782
Exp/Cntr=0.3,0.1

Type RM Length L Ch R = 1,12664,324,324,324
BEGIN DESCRIPTION:
Mapping XS 6552df5f
END DESCRIPTION:
XS GIS Cut Line= 3
      1692681.28      7039097.24      1692911.77      7039295.17
      1693532.83      7039853.74
#Sta/Elev= 30
  4698.4 1570.96  4794.2 1558.41  4811.0 1553.52  4835.9 1546.32  4878.7 1537.93
  4904.2 1530.18  4928.0 1522.67  4985.1 1508.00  4992.8 1505.40  5002.2 1496.62
  5007.7 1496.62  5013.6 1492.80  5023.4 1489.96  5023.9 1489.46  5032.2 1489.96
  5048.7 1493.97  5070.4 1496.41  5113.0 1495.84  5119.7 1493.25  5127.2 1493.69
  5133.9 1495.85  5154.0 1497.37  5211.7 1497.45  5225.9 1499.17  5374.6 1500.18
  5480.7 1505.13  5523.4 1508.80  5622.8 1512.16  5693.0 1518.83  5837.5 1524.16
#Mann=6,-1,0
  4698.4    0.07       0  4811.0   0.035       0  4904.2    0.07       0
  5023.4    0.07       0  5032.2    0.07       0  5154.0   0.035       0
Bank Sta=5023.4,5032.2
Exp/Cntr=0.3,0.1

Type RM Length L Ch R = 1,12340,329,329,329
BEGIN DESCRIPTION:
Mapping XS a04db3af
END DESCRIPTION:
XS GIS Cut Line= 3
      1692514.17      7039385.00      1692801.96      7039585.54
      1693645.68      7039995.68
#Sta/Elev= 30
  4649.7 1549.20  4660.3 1549.04  4687.3 1543.85  4746.6 1537.62  4760.4 1534.08
  4767.6 1533.68  4773.7 1530.04  4782.4 1530.25  4788.5 1526.63  4803.3 1529.17
  4809.4 1526.51  4818.2 1526.83  4854.0 1522.63  4860.1 1520.53  4904.6 1516.31
  4918.9 1513.50  4946.4 1505.03  4961.3 1498.73  4967.6 1492.40  4976.1 1488.13
  4986.5 1486.39  4987.0 1485.89  4995.4 1486.39  5081.1 1493.88  5237.3 1496.00
  5408.0 1504.64  5447.6 1508.03  5537.6 1510.81  5678.7 1520.84  5938.6 1529.29
#Mann=3,-1,0
  4649.7   0.035       0  4986.5   0.035       0  4995.4   0.035       0
Bank Sta=4986.5,4995.4
Exp/Cntr=0.3,0.1

Type RM Length L Ch R = 1,12011,321,321,321
BEGIN DESCRIPTION:
Mapping XS 120be95b
END DESCRIPTION:
XS GIS Cut Line= 3
      1692474.70      7039782.15      1692705.17      7039883.71
      1693439.57      7040056.90
#Sta/Elev= 30
  4751.0 1536.54  4755.0 1535.28  4795.0 1531.87  4824.9 1524.36  4838.8 1522.66
  4882.5 1514.11  4893.4 1513.28  4923.7 1506.14  4929.2 1505.62  4947.0 1500.16
  4952.5 1499.33  4969.9 1488.76  4971.4 1483.62  4971.9 1483.12  4980.3 1483.62
  5005.3 1484.57  5013.0 1487.31  5023.2 1488.48  5074.6 1491.43  5156.8 1490.84
  5197.9 1491.57  5269.8 1497.22  5372.6 1502.03  5432.3 1506.04  5547.2 1509.63
  5578.0 1511.61  5639.7 1517.92  5654.2 1518.00  5732.2 1522.29  5757.4 1522.67
#Mann=3,-1,0
  4751.0   0.035       0  4971.4   0.035       0  4980.3   0.035       0
Bank Sta=4971.4,4980.3
Exp/Cntr=0.3,0.1

Type RM Length L Ch R = 1,11690,381,381,381
BEGIN DESCRIPTION:
Mapping XS 1e18ec9a
END DESCRIPTION:
XS GIS Cut Line= 3
      1692266.38      7040161.49      1692655.26      7040187.53
      1693588.56      7040243.05
#Sta/Elev= 30
  4610.6 1548.01  4639.3 1544.30  4769.6 1535.45  4783.7 1533.76  4829.7 1523.23
  4879.8 1516.14  4899.9 1514.28  4933.7 1506.39  4960.0 1498.57  4980.0 1489.14
  4993.3 1481.67  4993.8 1481.17  5002.2 1481.67  5010.1 1481.68  5020.1 1483.65
  5040.2 1485.13  5060.2 1484.27  5088.8 1487.79  5160.4 1488.77  5427.6 1499.36
  5440.9 1499.03  5521.0 1502.35  5551.1 1505.13  5631.2 1507.43  5751.4 1514.98
  5766.3 1514.81  5801.5 1517.09  5901.7 1520.91  5930.6 1523.30  5935.3 1522.85
#Mann=3,-1,0
  4610.6   0.035       0  4993.3   0.035       0  5002.2   0.035       0
Bank Sta=4993.3,5002.2
Exp/Cntr=0.3,0.1

Type RM Length L Ch R = 1,11309,333,333,333
BEGIN DESCRIPTION:
Mapping XS 563af087
END DESCRIPTION:
XS GIS Cut Line= 3
      1692302.62      7040637.41      1692757.45      7040536.72
      1693491.77      7040399.91
#Sta/Elev= 30
  4532.6 1524.57  4595.3 1523.28  4600.4 1524.12  4709.2 1519.95  4736.4 1516.03
  4741.5 1516.46  4770.6 1512.28  4785.2 1511.71  4828.8 1506.51  4833.9 1507.95
  4872.4 1503.66  4877.5 1504.41  4921.1 1495.79  4926.3 1495.69  4955.0 1483.10
  4985.7 1481.60  4990.1 1478.84  4990.6 1478.34  4999.1 1478.84  5006.1 1481.21
  5015.0 1481.89  5077.9 1484.12  5097.7 1483.28  5372.3 1499.27  5404.4 1502.64
  5474.0 1506.02  5515.0 1512.43  5555.4 1515.36  5615.3 1518.17  5745.4 1521.61
#Mann=3,-1,0
  4532.6   0.035       0  4990.1   0.035       0  4999.1   0.035       0
Bank Sta=4990.1,4999.1
Exp/Cntr=0.3,0.1

Type RM Length L Ch R = 1,10976,273,273,273
BEGIN DESCRIPTION:
Mapping XS 74d21ab8
END DESCRIPTION:
XS GIS Cut Line= 3
      1692370.26      7040830.13      1692953.64      7040781.51
      1693467.53      7040727.69
#Sta/Elev= 30
  4412.7 1513.94  4477.7 1509.23  4537.9 1500.97  4621.1 1499.99  4668.3 1498.34
  4736.5 1491.45  4741.5 1491.86  4788.7 1484.05  4838.9 1479.75  4848.9 1479.21
  4879.0 1481.05  4909.2 1480.78  4977.3 1477.84  4977.8 1476.63  4978.3 1476.13
  4986.9 1476.63  4989.4 1477.78  5001.3 1478.90  5029.6 1484.22  5049.7 1486.42
  5077.4 1492.72  5082.4 1492.86  5090.0 1495.24  5120.1 1500.47  5150.3 1502.85
  5175.6 1506.91  5220.7 1511.85  5268.9 1515.29  5331.3 1517.90  5514.8 1522.73
#Mann=3,-1,0
  4412.7   0.035       0  4977.8   0.035       0  4986.9   0.035       0
Bank Sta=4977.8,4986.9
Exp/Cntr=0.3,0.1

Type RM Length L Ch R = 1,10703,489,489,489
BEGIN DESCRIPTION:
Mapping XS 76dcbb37
END DESCRIPTION:
XS GIS Cut Line= 3
      1692463.49      7041079.22      1692912.75      7041040.15
      1693401.20      7040975.20
#Sta/Elev= 30
  4548.9 1509.19  4580.5 1507.89  4650.8 1500.86  4701.0 1498.46  4751.2 1494.42
  4791.3 1489.42  4821.4 1484.34  4849.0 1481.50  4881.7 1480.25  4972.0 1479.22
  4993.9 1473.39  4994.4 1472.89  5003.0 1473.39  5032.4 1475.20  5042.5 1474.38
  5050.8 1477.67  5055.9 1477.97  5062.6 1479.95  5092.9 1480.97  5113.1 1483.17
  5123.2 1486.54  5129.1 1489.74  5134.1 1490.03  5153.4 1496.92  5163.5 1499.39
  5173.6 1500.47  5202.3 1506.05  5244.2 1510.91  5304.8 1514.57  5492.6 1517.65
#Mann=3,-1,0
  4548.9   0.035       0  4993.9   0.035       0  5003.0   0.035       0
Bank Sta=4993.9,5003
Exp/Cntr=0.3,0.1

Type RM Length L Ch R = 1,10214,260,260,260
BEGIN DESCRIPTION:
Mapping XS 0db769be
END DESCRIPTION:
XS GIS Cut Line= 3
      1692443.14      7041160.97      1692864.12      7041479.97
      1693287.30      7041723.02
#Sta/Elev= 30
  4471.7 1508.55  4492.2 1507.75  4556.7 1500.10  4606.6 1497.67  4642.0 1494.09
  4741.9 1487.36  4771.0 1483.25  4812.8 1480.71  4977.0 1476.24  4991.5 1474.69
  4997.3 1472.05  5002.9 1472.05  5012.4 1468.93  5017.6 1468.63  5018.1 1468.13
  5026.7 1468.63  5027.9 1470.66  5043.7 1472.41  5093.2 1473.70  5116.2 1481.92
  5151.6 1488.95  5183.2 1490.72  5188.9 1493.28  5220.0 1496.21  5269.5 1505.12
  5350.0 1511.27  5371.5 1514.66  5446.3 1519.42  5473.7 1524.24  5487.9 1525.44
#Mann=3,-1,0
  4471.7   0.035       0  5017.6   0.035       0  5026.7   0.035       0
Bank Sta=5017.6,5026.7
Exp/Cntr=0.3,0.1

Type RM Length L Ch R = 1,9954,341,341,341
BEGIN DESCRIPTION:
Mapping XS 830d6624
END DESCRIPTION:
XS GIS Cut Line= 3
      1692382.34      7041308.51      1692749.10      7041696.98
      1693014.91      7041954.15
#Sta/Elev= 30
  4467.9 1507.26  4497.6 1505.91  4561.5 1497.82  4604.0 1495.20  4625.0 1492.42
  4724.2 1485.00  4787.7 1478.02  4978.6 1472.19  4992.8 1470.84  4999.4 1469.12
  5037.7 1466.92  5038.2 1466.42  5047.0 1466.92  5063.7 1476.39  5070.7 1478.66
  5077.8 1482.31  5084.8 1482.47  5092.0 1485.63  5098.9 1485.24  5106.1 1488.21
  5113.1 1488.53  5120.3 1491.76  5141.4 1494.15  5183.8 1503.00  5233.2 1507.61
  5261.5 1511.55  5311.2 1516.76  5332.3 1522.12  5360.6 1527.72  5372.0 1528.95
#Mann=3,-1,0
  4467.9   0.035       0  5037.7   0.035       0  5047.0   0.035       0
Bank Sta=5037.7,5047
Exp/Cntr=0.3,0.1

Type RM Length L Ch R = 1,9613,278,278,278
BEGIN DESCRIPTION:
Mapping XS e41a628f
END DESCRIPTION:
XS GIS Cut Line= 3
      1692365.00      7041447.45      1692506.05      7041940.04
      1692885.80      7042196.10
#Sta/Elev= 30
  4493.9 1499.45  4516.3 1496.51  4577.7 1494.07  4702.5 1478.90  4754.5 1474.09
  4913.7 1470.79  4947.5 1466.61  5008.7 1466.56  5021.6 1463.60  5022.1 1463.10
  5030.9 1463.60  5032.3 1468.88  5047.3 1471.48  5077.2 1480.87  5125.6 1489.58
  5170.2 1495.36  5257.1 1503.63  5299.1 1505.17  5314.1 1507.79  5320.2 1506.79
  5329.1 1509.08  5335.1 1507.80  5350.1 1510.62  5371.1 1510.06  5386.1 1512.79
  5407.1 1513.28  5437.0 1517.56  5443.1 1516.83  5458.0 1521.38  5464.3 1520.81
#Mann=3,-1,0
  4493.9   0.035       0  5021.6   0.035       0  5030.9   0.035       0
Bank Sta=5021.6,5030.9
Exp/Cntr=0.3,0.1

Type RM Length L Ch R = 1,9335,321,321,321
BEGIN DESCRIPTION:
Mapping XS 77db704d
END DESCRIPTION:
XS GIS Cut Line= 3
      1692227.38      7041578.45      1692242.57      7041988.65
      1692265.36      7042281.58
#Sta/Elev= 30
  4590.1 1490.40  4599.7 1488.95  4662.8 1485.27  4679.7 1483.81  4699.7 1481.64
  4759.8 1472.02  4769.8 1471.26  4789.8 1470.15  4839.8 1469.34  4933.0 1469.31
  4969.9 1468.43  4979.9 1466.90  4992.9 1461.00  4993.4 1460.50  5002.2 1460.50
  5002.7 1461.00  5010.0 1461.96  5020.0 1464.88  5030.0 1465.21  5060.1 1467.77
  5070.1 1467.74  5080.2 1469.42  5090.2 1472.82  5095.8 1476.67  5150.4 1480.81
  5210.6 1488.51  5225.5 1488.76  5250.7 1490.41  5290.1 1494.56  5294.4 1494.56
#Mann=3,-1,0
  4590.1   0.035       0  4992.9   0.035       0  5002.7   0.035       0
Bank Sta=4992.9,5002.7
Exp/Cntr=0.3,0.1

Type RM Length L Ch R = 1,9014,276,276,276
BEGIN DESCRIPTION:
Mapping XS 02f2c320
END DESCRIPTION:
XS GIS Cut Line= 3
      1692144.91      7041565.50      1691936.59      7042040.73
      1691821.59      7042322.80
#Sta/Elev= 30
  4483.8 1486.92  4563.0 1482.76  4621.8 1478.39  4639.4 1476.76  4668.5 1471.72
  4674.0 1471.79  4691.9 1469.00  4744.1 1467.30  4803.2 1467.16  4879.6 1465.51
  4934.2 1465.88  4947.5 1465.08  4965.4 1461.49  4988.8 1462.28  5018.5 1460.04
  5019.0 1459.54  5028.4 1460.04  5042.1 1467.32  5047.5 1468.43  5053.7 1474.73
  5064.5 1478.55  5071.5 1480.73  5095.6 1484.58  5107.7 1487.47  5125.0 1488.79
  5183.9 1495.87  5215.7 1497.85  5256.0 1498.17  5285.5 1500.78  5307.3 1501.47
#Mann=3,-1,0
  4483.8   0.035       0  5018.5   0.035       0  5028.4   0.035       0
Bank Sta=5018.5,5028.4
Exp/Cntr=0.3,0.1

Type RM Length L Ch R = 1,8738,230,230,230
BEGIN DESCRIPTION:
Mapping XS 97a43784
END DESCRIPTION:
XS GIS Cut Line= 3
      1692112.39      7041503.60      1691714.15      7041952.84
      1691521.50      7042213.67
#Sta/Elev= 30
  4403.4 1487.12  4468.4 1482.09  4539.5 1478.79  4588.8 1474.69  4617.2 1473.36
  4801.2 1465.99  4900.8 1464.16  4950.1 1461.82  4964.3 1462.41  4980.3 1458.18
  4980.8 1457.68  4990.2 1458.18  4992.8 1459.76  4999.3 1460.50  5013.5 1459.54
  5035.0 1460.96  5063.7 1459.33  5078.3 1461.03  5084.8 1462.33  5099.1 1468.63
  5113.8 1473.46  5128.4 1476.97  5134.6 1479.67  5143.0 1480.91  5163.9 1486.41
  5178.5 1488.79  5184.7 1490.68  5214.0 1495.10  5234.8 1497.05  5328.0 1500.99
#Mann=3,-1,0
  4403.4   0.035       0  4980.3   0.035       0  4990.2   0.035       0
Bank Sta=4980.3,4990.2
Exp/Cntr=0.3,0.1

Type RM Length L Ch R = 1,8508,218,218,218
BEGIN DESCRIPTION:
Mapping XS 92cb296b
END DESCRIPTION:
XS GIS Cut Line= 3
      1691969.67      7041391.76      1691534.53      7041821.47
      1691372.87      7042036.29
#Sta/Elev= 30
  4391.6 1487.49  4420.5 1484.99  4427.6 1483.75  4477.1 1480.28  4519.5 1476.09
  4576.1 1472.69  4774.1 1464.97  4958.0 1460.46  4979.1 1458.32  4986.3 1456.40
  5003.2 1456.93  5007.9 1455.82  5009.2 1453.77  5009.7 1453.27  5019.1 1453.77
  5036.3 1458.94  5043.3 1459.23  5072.4 1455.97  5078.7 1457.67  5093.3 1466.65
  5099.5 1471.67  5107.8 1476.41  5114.1 1481.38  5122.4 1485.33  5128.7 1487.86
  5157.8 1494.38  5172.4 1495.64  5178.6 1495.24  5193.2 1496.07  5272.0 1497.11
#Mann=3,-1,0
  4391.6   0.035       0  5009.2   0.035       0  5019.1   0.035       0
Bank Sta=5009.2,5019.1
Exp/Cntr=0.3,0.1

Type RM Length L Ch R = 1,8290,188,188,188
BEGIN DESCRIPTION:
Mapping XS 5e2fa1ff
END DESCRIPTION:
XS GIS Cut Line= 3
      1691926.23      7041219.27      1691362.00      7041698.86
      1691315.46      7041903.42
#Sta/Elev= 30
  4262.2 1497.19  4283.4 1495.61  4312.0 1490.76  4361.4 1485.69  4375.7 1483.17
  4432.8 1477.04  4468.0 1474.45  4730.4 1464.14  4915.0 1458.77  4929.2 1457.98
  4943.5 1455.36  4957.8 1454.07  4964.4 1454.65  4985.7 1453.72  4998.2 1456.49
  5004.8 1456.49  5017.4 1453.53  5017.9 1453.03  5027.3 1453.53  5042.8 1456.53
  5052.4 1460.49  5063.4 1470.57  5073.6 1476.18  5083.9 1479.97  5094.1 1482.40
  5100.6 1483.19  5148.8 1482.92  5191.8 1484.35  5196.9 1483.53  5212.5 1484.69
#Mann=3,-1,0
  4262.2   0.035       0  5017.4   0.035       0  5027.3   0.035       0
Bank Sta=5017.4,5027.3
Exp/Cntr=0.3,0.1
