HEC-RAS study Clear Fork Brazos Rv.prj: Clear Fork Brazos Rv Base Level Engineering

--- Clear Fork Brazos Rv.g01 (geometry) --- (continued)

Type RM Length L Ch R = 1,1077959,683,683,683
BEGIN DESCRIPTION:
Mapping XS 7665d5bb
END DESCRIPTION:
XS GIS Cut Line= 2
      1299186.60      6947654.93      1298339.11      6946506.97
#Sta/Elev= 30
  4217.4 2160.98  4224.9 2161.21  4357.1 2162.74  4416.2 2163.36  4474.6 2165.20
  4702.3 2165.82  4773.2 2167.23  4796.3 2165.25  4817.1 2160.84  4867.2 2159.95
  4888.1 2158.28  4946.6 2156.92  4952.8 2154.98  4959.4 2155.12  4973.7 2152.11
  4982.1 2151.47  4988.3 2148.32  4994.6 2143.55  4996.6 2141.55  5012.6 2141.55
  5014.6 2143.55  5023.8 2148.93  5032.2 2156.69  5067.7 2164.03  5073.9 2166.22
  5145.8 2166.43  5153.3 2167.15  5182.6 2166.31  5295.2 2166.30  5644.3 2168.00
#Mann=5,-1,0
  4217.4    0.05       0  4224.9    0.12       0  4357.1    0.05       0
  4994.6    0.05       0  5014.6    0.05       0
Bank Sta=4994.6,5014.6
Exp/Cntr=0.3,0.1

Type RM Length L Ch R = 1,1077276,137,137,137
BEGIN DESCRIPTION:
Mapping XS 839c7847
END DESCRIPTION:
XS GIS Cut Line= 2
      1299194.67      6947595.35      1299393.97      6946891.42
#Sta/Elev= 30
  4525.1 2161.26  4678.2 2163.62  4731.8 2163.53  4799.7 2165.31  4823.7 2164.85
  4838.8 2162.83  4844.5 2161.13  4854.9 2160.37  4878.0 2159.43  4906.7 2160.30
  4927.7 2157.95  4951.1 2156.94  4969.2 2153.51  4985.0 2146.61  4990.2 2146.00
  4995.4 2141.83  4997.4 2139.83  5013.4 2139.83  5015.4 2141.83  5018.9 2144.86
  5024.1 2145.11  5031.6 2153.79  5058.1 2163.10  5063.3 2161.65  5073.2 2163.66
  5083.6 2164.18  5131.2 2163.14  5145.9 2161.94  5197.9 2165.32  5256.7 2165.46
#Mann=3,-1,0
  4525.1    0.05       0  4995.4    0.05       0  5015.4    0.05       0
Bank Sta=4995.4,5015.4
Exp/Cntr=0.3,0.1

Type RM Length L Ch R = 1,1077139,918,918,918
BEGIN DESCRIPTION:
Mapping XS 75dd4362
END DESCRIPTION:
XS GIS Cut Line= 2
      1299373.20      6947578.30      1299513.46      6946847.24
#Sta/Elev= 30
  4590.2 2160.86  4804.3 2164.60  4834.2 2161.15  4839.3 2161.60  4855.3 2159.94
  4967.3 2155.42  4987.6 2149.67  4995.3 2146.51  5000.3 2145.85  5005.0 2141.55
  5007.4 2139.55  5026.6 2139.55  5029.0 2141.55  5038.5 2145.97  5047.2 2151.39
  5058.9 2154.69  5099.2 2157.63  5109.8 2155.70  5120.0 2155.23  5150.5 2159.48
  5170.9 2158.99  5181.1 2160.21  5201.5 2159.60  5213.4 2157.83  5242.2 2157.91
  5252.4 2158.77  5260.3 2161.31  5265.4 2161.10  5272.7 2163.19  5334.6 2164.24
#Mann=3,-1,0
  4590.2    0.05       0  5005.0    0.03       0  5029.0    0.05       0
Bank Sta=5005,5029
Exp/Cntr=0.3,0.1

Type RM Length L Ch R = 1,1076221,1175,1175,1175
BEGIN DESCRIPTION:
Mapping XS 7752ce69
END DESCRIPTION:
XS GIS Cut Line= 2
      1300040.67      6947574.21      1299941.63      6946802.44
#Sta/Elev= 30
  4407.6 2159.09  4415.9 2159.53  4444.1 2159.37  4484.4 2159.96  4490.4 2160.49
  4534.8 2160.64  4615.5 2158.65  4676.0 2159.84  4797.0 2160.03  4847.4 2160.43
  4877.6 2161.22  4897.8 2160.84  4938.1 2161.01  4948.2 2159.55  4958.0 2155.43
  4963.1 2156.36  4968.4 2152.16  4988.5 2145.38  4998.6 2143.28  5008.7 2140.49
  5014.1 2139.67  5017.3 2137.67  5042.9 2137.67  5046.1 2139.67  5059.1 2141.82
  5069.2 2148.93  5079.3 2160.32  5089.4 2162.57  5159.9 2163.18  5185.7 2162.97
#Mann=3,-1,0
  4407.6    0.05       0  5014.1    0.05       0  5046.1    0.05       0
Bank Sta=5014.1,5046.1
Exp/Cntr=0.3,0.1

Type RM Length L Ch R = 1,1075046,1286,1286,1286
BEGIN DESCRIPTION:
Mapping XS e2d2d8aa
END DESCRIPTION:
XS GIS Cut Line= 2
      1300574.49      6947675.91      1300887.95      6945812.09
#Sta/Elev= 30
  4025.5 2155.13  4571.0 2158.51  4659.4 2151.28  4841.1 2154.49  4846.2 2151.69
  4865.0 2149.95  4946.2 2149.18  4962.3 2143.94  4967.3 2144.35  4978.9 2137.91
  4982.9 2135.91  5020.8 2135.91  5024.8 2137.91  5037.4 2140.34  5047.6 2148.47
  5057.7 2153.28  5088.5 2153.54  5128.7 2157.32  5144.0 2161.83  5149.0 2160.44
  5169.3 2164.18  5311.2 2168.61  5514.0 2167.79  5585.0 2169.37  5689.1 2177.14
  5716.8 2185.17  5757.4 2191.76  5805.1 2209.16  5858.8 2212.65  5915.5 2208.83
#Mann=3,-1,0
  4025.5    0.05       0  4978.9    0.05       0  5024.8    0.05       0
Bank Sta=4978.9,5024.8
Exp/Cntr=0.3,0.1

Type RM Length L Ch R = 1,1073760,859,859,859
BEGIN DESCRIPTION:
Mapping XS 37546d94
END DESCRIPTION:
XS GIS Cut Line= 3
      1301086.23      6948091.74      1301502.89      6947206.34
      1301320.68      6946182.47
#Sta/Elev= 30
  4452.2 2150.57  4905.6 2151.41  4911.1 2150.38  4920.5 2145.90  4928.4 2136.33
  4933.9 2131.31  4937.7 2131.81  4940.5 2130.81  4967.0 2130.81  4969.8 2131.81
  4974.0 2135.80  5008.9 2139.02  5047.9 2141.16  5064.2 2140.49  5086.3 2145.02
  5116.3 2146.82  5309.7 2146.78  5332.5 2149.54  5340.5 2151.84  5355.3 2153.24
  5459.5 2151.83  5530.6 2153.03  5730.7 2151.54  5967.4 2153.54  6089.3 2152.07
  6099.4 2150.19  6109.6 2152.39  6150.2 2154.59  6292.4 2156.72  6470.7 2161.88
#Mann=3,-1,0
  4452.2    0.05       0  4937.7    0.05       0  4969.8    0.05       0
Bank Sta=4937.7,4969.8
Exp/Cntr=0.3,0.1

Type RM Length L Ch R = 1,1072901,897,897,897
BEGIN DESCRIPTION:
Mapping XS b0865815
END DESCRIPTION:
XS GIS Cut Line= 3
      1301570.75      6948226.35      1302137.92      6947725.90
      1301596.42      6946401.31
#Sta/Elev= 30
  3874.2 2148.67  4527.9 2149.03  4837.8 2151.66  4885.8 2144.83  4930.8 2144.05
  4952.4 2142.05  4984.8 2132.50  4988.6 2129.60  4990.6 2127.60  5009.5 2127.60
  5011.5 2129.60  5016.7 2132.65  5022.1 2133.58  5028.1 2138.24  5038.9 2142.71
  5128.9 2147.63  5337.3 2143.76  5406.2 2145.44  5449.6 2151.44  5473.6 2151.48
  5492.2 2153.54  5521.6 2151.48  5535.8 2148.94  5589.8 2147.34  5676.3 2148.60
  5719.5 2151.60  5795.1 2149.48  5836.8 2150.66  5903.1 2149.51  6061.6 2154.26
#Mann=3,-1,0
  3874.2    0.05       0  4988.6    0.05       0  5011.5    0.05       0
Bank Sta=4988.6,5011.5
Exp/Cntr=0.3,0.1

Type RM Length L Ch R = 1,1072004,933,933,933
BEGIN DESCRIPTION:
Mapping XS f71df4c9
END DESCRIPTION:
XS GIS Cut Line= 2
      1301289.59      6948806.03      1302879.60      6947272.55
#Sta/Elev= 30
  2901.0 2150.04  3370.1 2148.39  3490.5 2146.29  3745.0 2148.30  4112.8 2147.58
  4360.3 2149.11  4650.2 2149.32  4714.0 2148.43  4721.0 2149.28  4742.3 2148.20
  4805.9 2148.17  4848.3 2142.51  4883.6 2142.20  4904.9 2140.55  4926.0 2140.95
  4933.2 2138.26  4940.2 2137.11  4954.3 2138.07  4982.6 2132.66  4996.8 2131.46
  4997.2 2127.24  4999.2 2125.24  5019.0 2125.24  5021.0 2127.24  5025.1 2127.36
  5032.3 2131.98  5039.2 2134.56  5053.4 2145.15  5060.6 2147.54  5110.0 2146.58
#Mann=3,-1,0
  2901.0    0.05       0  4997.2    0.05       0  5021.0    0.05       0
Bank Sta=4997.2,5021
Exp/Cntr=0.3,0.1

Type RM Length L Ch R = 1,1071071,835,835,835
BEGIN DESCRIPTION:
Mapping XS d5739eb3
END DESCRIPTION:
XS GIS Cut Line= 3
      1302153.96      6948517.07      1302544.56      6948091.75
      1303456.04      6948109.11
#Sta/Elev= 30
  3862.3 2147.46  4308.5 2146.12  4350.5 2146.73  4393.0 2146.29  4414.6 2147.14
  4530.2 2146.33  4560.2 2146.95  4650.2 2145.94  4720.3 2140.98  4770.3 2139.35
  4820.3 2139.99  4850.3 2141.83  4870.3 2141.79  4910.3 2139.62  4970.3 2138.36
  4990.3 2129.88  4998.0 2125.17  5000.4 2123.17  5024.1 2123.17  5026.5 2125.17
  5027.8 2127.91  5040.3 2128.53  5050.3 2130.10  5080.3 2138.25  5090.3 2142.97
  5100.3 2144.61  5130.3 2145.59  5170.3 2145.76  5240.3 2145.06  5351.4 2145.30
#Mann=3,-1,0
  3862.3    0.05       0  4998.0    0.03       0  5026.5    0.05       0
Bank Sta=4998,5026.5
Exp/Cntr=0.3,0.1

Type RM Length L Ch R = 1,1070236,1261,1261,1261
BEGIN DESCRIPTION:
Mapping XS 48e021f8
END DESCRIPTION:
XS GIS Cut Line= 2
      1301940.59      6949739.23      1303694.46      6948224.24
#Sta/Elev= 30
  3621.8 2146.33  3852.3 2151.92  3874.1 2151.08  3952.0 2151.87  4058.4 2151.57
  4093.5 2149.53  4150.5 2148.96  4355.7 2142.60  4504.8 2141.59  4576.1 2142.94
  4618.7 2145.28  4859.2 2145.21  4873.4 2144.42  4909.4 2139.41  4930.4 2140.80
  4944.7 2136.66  4951.3 2130.61  4958.9 2127.11  4973.2 2123.23  4983.8 2122.32
  4988.2 2121.32  5031.8 2121.32  5036.2 2122.32  5057.7 2136.84  5079.6 2136.52
  5114.7 2138.36  5135.6 2142.25  5149.8 2143.32  5341.8 2144.45  5939.4 2142.86
#Mann=3,-1,0
  3621.8    0.05       0  4983.8    0.05       0  5036.2    0.05       0
Bank Sta=4983.8,5036.2
Exp/Cntr=0.3,0.1

Type RM Length L Ch R = 1,1068975,746,746,746
BEGIN DESCRIPTION:
Mapping XS 289b88c4
END DESCRIPTION:
XS GIS Cut Line= 3
      1303030.43      6949385.82      1303956.33      6949410.85
      1304439.04      6948761.68
#Sta/Elev= 30
  3751.4 2141.77  3846.0 2146.61  4019.0 2142.06  4186.1 2146.78  4296.2 2147.91
  4526.3 2141.90  4656.3 2141.55  4771.1 2143.32  4785.7 2142.65  4800.3 2139.50
  4829.6 2136.87  4850.4 2135.20  4856.6 2135.94  4879.6 2131.72  4935.9 2130.15
  4956.7 2131.08  4971.4 2126.29  4979.7 2121.94  4985.7 2121.43  4988.1 2119.43
  5011.9 2119.43  5014.3 2121.43  5021.4 2121.54  5029.8 2124.62  5042.6 2132.39
  5050.6 2132.19  5056.9 2133.71  5165.4 2134.34  5221.7 2140.55  5486.6 2138.39
#Mann=3,-1,0
  3751.4    0.05       0  4985.7    0.05       0  5014.3    0.05       0
Bank Sta=4985.7,5014.3
Exp/Cntr=0.3,0.1

Type RM Length L Ch R = 1,1068229,694,694,694
BEGIN DESCRIPTION:
Mapping XS 91102b93
END DESCRIPTION:
XS GIS Cut Line= 2
      1302884.66      6949457.10      1304660.54      6949652.53
#Sta/Elev= 30
  3369.1 2141.92  3389.6 2142.78  3409.7 2141.25  3423.9 2141.78  3429.8 2140.60
  3514.9 2139.19  3580.7 2143.25  3661.2 2143.94  3822.2 2140.82  4113.9 2141.98
  4254.8 2138.05  4345.3 2136.89  4747.7 2138.18  4793.6 2136.78  4838.3 2130.49
  4948.9 2131.53  4959.0 2128.30  4969.0 2122.42  4975.6 2120.39  4980.6 2120.33
  4987.7 2117.27  4989.7 2115.27  5009.5 2115.27  5011.5 2117.27  5019.3 2122.76
  5039.5 2125.41  5059.6 2130.48  5071.6 2130.69  5089.8 2136.55  5155.7 2135.75
#Mann=3,-1,0
  3369.1    0.05       0  4987.7    0.05       0  5011.5    0.05       0
Bank Sta=4987.7,5011.5
Exp/Cntr=0.3,0.1

Type RM Length L Ch R = 1,1067535,1145,1145,1145
BEGIN DESCRIPTION:
Mapping XS b8860d5e
END DESCRIPTION:
XS GIS Cut Line= 4
      1303074.44      6949709.65      1303760.68      6949802.93
      1304200.40      6950216.00      1304420.17      6950109.45
#Sta/Elev= 30
  3826.8 2138.56  3877.8 2139.35  3898.0 2138.94  3988.8 2139.20  4002.1 2138.65
  4039.3 2138.96  4241.1 2137.23  4463.2 2136.58  4589.8 2134.83  4731.1 2135.97
  4738.2 2135.46  4745.1 2133.73  4752.4 2133.56  4759.3 2132.07  4780.7 2130.04
  4950.6 2126.98  4957.5 2125.64  4971.7 2121.29  4986.5 2115.34  4988.1 2114.34
  5003.9 2114.34  5005.5 2115.34  5006.9 2120.80  5014.2 2124.08  5021.1 2128.15
  5049.4 2128.63  5063.5 2131.68  5070.8 2134.27  5085.0 2135.74  5366.9 2135.12
#Mann=3,-1,0
  3826.8    0.05       0  4986.5    0.05       0  5005.5    0.05       0
Bank Sta=4986.5,5005.5
Exp/Cntr=0.3,0.1

Type RM Length L Ch R = 1,1066390,1232,1232,1232
BEGIN DESCRIPTION:
Mapping XS 958c2027
END DESCRIPTION:
XS GIS Cut Line= 3
      1303074.09      6951164.66      1303950.81      6950383.42
      1304419.58      6950149.03
#Sta/Elev= 30
  4140.1 2140.99  4492.3 2134.24  4620.2 2129.98  4626.9 2128.07  4634.4 2129.68
  4641.1 2127.52  4648.6 2130.20  4662.8 2130.78  4733.1 2126.78  4761.5 2129.64
  4797.5 2129.70  4832.6 2127.70  4861.0 2123.67  4867.7 2120.73  4903.6 2119.78
  4917.9 2121.57  4924.5 2119.01  4931.6 2123.47  4938.8 2123.58  4959.7 2117.85
  4985.5 2116.00  4987.5 2114.00  5008.1 2114.00  5010.1 2116.00  5016.5 2119.04
  5059.2 2124.26  5116.0 2122.07  5165.3 2132.01  5193.8 2133.34  5838.5 2135.14
#Mann=3,-1,0
  4140.1    0.05       0  4985.5    0.05       0  5010.1    0.05       0
Bank Sta=4985.5,5010.1
Exp/Cntr=0.3,0.1

Type RM Length L Ch R = 1,1065158,416,416,416
BEGIN DESCRIPTION:
Mapping XS 9e2504b2
END DESCRIPTION:
XS GIS Cut Line= 3
      1304492.04      6951397.50      1304832.97      6950898.11
      1305116.20      6950542.87
#Sta/Elev= 30
  4383.3 2133.92  4500.8 2132.68  4536.7 2131.24  4614.5 2123.77  4650.4 2122.38
  4773.0 2122.14  4830.7 2123.62  4867.0 2120.00  4874.7 2115.79  4880.7 2117.12
  4889.6 2121.56  4952.5 2121.21  4961.4 2119.73  4976.0 2114.09  4979.6 2111.39
  4981.6 2109.39  5002.2 2109.39  5004.2 2111.39  5017.7 2118.73  5032.1 2121.56
  5046.5 2122.30  5110.6 2121.46  5117.0 2119.31  5139.4 2116.90  5153.8 2120.31
  5181.0 2120.69  5189.0 2121.62  5217.9 2130.45  5238.7 2131.04  5442.3 2129.29
#Mann=3,-1,0
  4383.3    0.05       0  4979.6    0.05       0  5004.2    0.05       0
Bank Sta=4979.6,5004.2
Exp/Cntr=0.3,0.1

Type RM Length L Ch R = 1,1064742,1011,1011,1011
BEGIN DESCRIPTION:
Mapping XS 862a7fed
END DESCRIPTION:
XS GIS Cut Line= 2
      1304755.98      6951762.34      1305303.95      6950922.51
#Sta/Elev= 30
  4298.3 2145.15  4307.6 2145.57  4322.7 2144.07  4380.0 2142.55  4431.3 2139.31
  4554.2 2134.87  4690.8 2126.84  4711.8 2124.87  4793.0 2123.95  4814.5 2125.28
  4820.5 2124.79  4835.6 2126.48  4871.8 2126.20  4914.0 2118.48  4936.3 2119.89
  4959.4 2118.69  4980.4 2114.32  4985.7 2110.92  4987.7 2108.92  5008.8 2108.92
  5010.8 2110.92  5022.6 2117.78  5037.7 2120.25  5089.1 2121.50  5095.0 2122.23
  5103.5 2125.18  5139.3 2128.50  5175.1 2129.22  5197.7 2128.17  5301.1 2128.43
#Mann=3,-1,0
  4298.3    0.05       0  4985.7    0.05       0  5010.8    0.05       0
Bank Sta=4985.7,5010.8
Exp/Cntr=0.3,0.1

Type RM Length L Ch R = 1,1063731,1337,1337,1337
BEGIN DESCRIPTION:
Mapping XS 083b31eb
END DESCRIPTION:
XS GIS Cut Line= 2
      1306421.95      6952647.21      1305477.94      6950856.85
#Sta/Elev= 30
  3911.7 2172.30  4235.2 2176.29  4367.4 2172.26  4405.8 2173.54  4419.5 2170.78
  4427.8 2172.34  4433.5 2168.12  4449.8 2171.25  4455.5 2166.94  4471.9 2168.38
  4477.5 2163.47  4493.9 2163.96  4499.5 2160.40  4510.0 2160.22  4537.9 2153.81
  4840.6 2137.94  4923.1 2122.02  4961.5 2117.64  4996.1 2116.91  5005.5 2114.05
  5005.7 2109.33  5008.5 2108.33  5040.8 2109.33  5055.2 2109.24  5071.6 2114.94
  5077.3 2112.91  5093.6 2118.08  5165.7 2118.24  5278.7 2125.09  5935.7 2127.89
#Mann=3,-1,0
  3911.7    0.05       0  5005.7    0.05       0  5040.8    0.05       0
Bank Sta=5005.7,5040.8
Exp/Cntr=0.3,0.1

Type RM Length L Ch R = 1,1062394,838,838,838
BEGIN DESCRIPTION:
Mapping XS 12e07aba
END DESCRIPTION:
XS GIS Cut Line= 3
      1306965.32      6951455.20      1306299.09      6950649.07
      1305599.75      6950875.52
#Sta/Elev= 30
  3847.6 2149.20  4087.7 2137.21  4108.5 2137.49  4307.8 2129.79  4378.2 2129.71
  4392.5 2127.53  4449.8 2128.01  4499.3 2126.21  4584.0 2125.77  4740.3 2121.72
  4950.3 2120.66  4960.8 2119.57  4973.8 2114.08  4981.8 2112.97  4987.5 2104.83
  4989.5 2103.83  5010.6 2103.83  5012.6 2104.83  5013.3 2109.42  5032.6 2110.32
  5044.9 2113.51  5086.9 2115.77  5128.6 2113.55  5165.8 2115.56  5223.6 2115.75
  5261.8 2117.27  5318.2 2122.53  5538.9 2121.84  5587.0 2122.45  5628.5 2124.46
#Mann=3,-1,0
  3847.6    0.05       0  4987.5    0.05       0  5012.6    0.05       0
Bank Sta=4987.5,5012.6
Exp/Cntr=0.3,0.1

Type RM Length L Ch R = 1,1061556,920,920,920
BEGIN DESCRIPTION:
Clear Fork Brazos Rv 334.0
END DESCRIPTION:
XS GIS Cut Line= 3
      1307154.97      6951487.97      1305905.00      6950088.00
      1305705.01      6949538.03
#Sta/Elev= 30
  3123.2 2166.99  3179.6 2166.64  3264.9 2159.72  3300.0 2159.31  3470.5 2140.66
  3682.9 2130.67  4001.4 2123.02  4355.8 2119.72  4574.9 2120.09  4695.3 2113.53
  4844.1 2116.24  4957.8 2115.17  4972.0 2112.27  4987.4 2104.00  4989.4 2103.00
  5012.6 2104.00  5021.3 2109.57  5045.9 2113.23  5101.7 2111.99  5127.0 2113.67
  5132.3 2116.37  5149.0 2118.85  5170.2 2117.18  5180.9 2118.29  5188.2 2120.66
  5193.5 2124.92  5202.2 2126.71  5397.0 2126.87  5500.1 2131.97  5585.2 2140.95
#Mann=3,-1,0
  3123.2    0.05       0  4987.4    0.05       0  5012.6    0.05       0
Bank Sta=4987.4,5012.6
Exp/Cntr=0.3,0.1

Type RM Length L Ch R = 1,1060636,1286,1286,1286
BEGIN DESCRIPTION:
Mapping XS c933e62d
END DESCRIPTION:
XS GIS Cut Line= 4
      1307198.51      6951248.67      1306419.01      6950575.78
      1306645.54      6950029.45      1306079.63      6949483.52
#Sta/Elev= 30
  3654.7 2154.24  3672.3 2154.44  3678.9 2153.20  3693.2 2153.75  3699.8 2152.26
  3721.7 2151.18  3742.5 2148.34  3806.2 2142.92  4182.4 2125.98  4317.3 2124.43
  4494.0 2120.44  4703.7 2120.19  4822.9 2117.97  4894.5 2111.88  4985.2 2110.48
  4993.9 2102.42  4995.5 2101.42  5012.5 2101.42  5014.1 2102.42  5017.6 2105.30
  5039.3 2109.85  5060.9 2112.69  5125.7 2117.92  5131.1 2120.18  5136.7 2119.45
  5169.2 2122.75  5376.2 2122.15  5715.8 2124.65  5928.0 2124.60  6062.2 2126.69
#Mann=3,-1,0
  3654.7    0.05       0  4993.9    0.05       0  5014.1    0.05       0
Bank Sta=4993.9,5014.1
Exp/Cntr=0.3,0.1

Type RM Length L Ch R = 1,1059350,577,577,577
BEGIN DESCRIPTION:
Clear Fork Brazos Rv 333.0
END DESCRIPTION:
XS GIS Cut Line= 3
      1307704.99      6950587.96      1307605.00      6950188.00
      1306005.03      6949338.01
#Sta/Elev= 30
  4583.5 2139.06  4642.7 2132.61  4730.3 2127.00  4789.6 2119.50  4848.9 2116.75
  4854.0 2114.52  4903.0 2108.95  4972.6 2108.15  4994.6 2104.79  4997.8 2102.79
  5031.7 2102.79  5034.9 2104.79  5047.9 2108.17  5063.7 2109.05  5143.0 2107.76
  5165.6 2109.10  5179.8 2111.92  5218.1 2114.15  5233.6 2116.92  5366.3 2120.40
  5505.3 2116.73  5586.1 2118.79  5743.1 2115.74  5816.6 2116.76  5904.5 2121.47
  5970.4 2122.98  6615.0 2125.38  6711.4 2128.24  6771.7 2132.22  6807.5 2132.07
#Mann=3,-1,0
  4583.5    0.05       0  4994.6    0.03       0  5034.9    0.05       0
Bank Sta=4994.6,5034.9
Exp/Cntr=0.3,0.1

Type RM Length L Ch R = 1,1058773,553,553,553
BEGIN DESCRIPTION:
Clear Fork Brazos Rv 332.0
END DESCRIPTION:
XS GIS Cut Line= 3
      1308055.01      6950588.03      1307705.00      6949638.00
      1306905.03      6948888.03
#Sta/Elev= 30
  3988.7 2134.61  4244.5 2123.90  4317.6 2119.49  4322.9 2120.94  4348.0 2118.49
  4372.4 2120.22  4415.0 2117.44  4500.3 2116.55  4596.2 2109.38  4955.5 2106.68
  4969.2 2104.72  4979.4 2101.09  4981.8 2099.09  5007.7 2099.09  5010.1 2101.09
  5015.1 2104.07  5029.3 2105.22  5036.6 2110.10  5057.6 2119.32  5411.7 2120.64
  5461.0 2117.93  5503.5 2117.51  5637.9 2121.48  5779.5 2123.70  5899.7 2123.29
  5949.0 2124.98  5956.3 2123.44  5970.5 2123.35  6055.5 2126.83  6097.7 2131.60
#Mann=3,-1,0
  3988.7    0.05       0  4979.4    0.03       0  5010.1    0.05       0
Bank Sta=4979.4,5010.1
Exp/Cntr=0.3,0.1

Type RM Length L Ch R = 1,1058220,524,524,524
BEGIN DESCRIPTION:
Clear Fork Brazos Rv 331.0
END DESCRIPTION:
XS GIS Cut Line= 3
      1308105.00      6950487.95      1308105.00      6949738.00
      1307404.99      6948287.98
#Sta/Elev= 30
  4249.3 2131.64  4389.3 2123.41  4549.3 2118.64  4639.3 2118.34  4669.3 2115.39
  4759.3 2112.97  4809.3 2109.30  4919.3 2107.75  4959.3 2109.07  4969.3 2104.19
  4979.8 2101.08  4982.6 2099.08  5013.0 2099.08  5015.8 2101.08  5021.5 2105.72
  5053.0 2107.60  5154.7 2109.28  5216.8 2108.57  5232.4 2110.68  5239.4 2114.22
  5262.0 2118.56  5634.8 2120.09  5702.6 2119.38  5754.3 2120.81  5860.8 2120.59
  6165.8 2122.99  6324.0 2128.81  6398.4 2135.98  6459.7 2140.36  6609.4 2145.19
#Mann=3,-1,0
  4249.3    0.05       0  4979.8    0.05       0  5015.8    0.05       0
Bank Sta=4979.8,5015.8
Exp/Cntr=0.3,0.1

Type RM Length L Ch R = 1,1057696,616,616,616
BEGIN DESCRIPTION:
Clear Fork Brazos Rv 330.0
END DESCRIPTION:
XS GIS Cut Line= 3
      1308121.39      6950374.29      1308565.82      6949832.64
      1308855.00      6948338.00
#Sta/Elev= 30
  4395.3 2124.48  4693.6 2116.23  4829.2 2105.93  4856.5 2107.93  4893.0 2106.65
  4913.9 2103.53  4928.2 2103.92  4934.7 2101.58  4956.9 2100.86  4963.4 2096.44
  4965.8 2096.62  4969.4 2094.62  5008.5 2094.62  5012.1 2096.62  5020.8 2095.72
  5027.2 2103.40  5035.1 2101.23  5041.6 2106.29  5049.5 2105.79  5055.9 2111.01
  5070.3 2109.48  5076.8 2113.75  5084.6 2113.68  5091.1 2116.73  5272.3 2115.42
  6261.8 2115.86  6363.7 2117.23  6475.7 2121.55  6567.4 2127.24  6618.3 2127.06
#Mann=3,-1,0
  4395.3    0.05       0  4965.8    0.05       0  5012.1    0.05       0
Bank Sta=4965.8,5012.1
Exp/Cntr=0.3,0.1

Type RM Length L Ch R = 1,1057080,990,990,990
BEGIN DESCRIPTION:
Clear Fork Brazos Rv 329.0
END DESCRIPTION:
XS GIS Cut Line= 3
      1308505.02      6950587.98      1308905.00      6950188.00
      1308905.00      6949656.75
#Sta/Elev= 30
  4434.7 2134.38  4462.9 2132.15  4477.1 2132.03  4519.5 2128.60  4533.7 2128.42
  4590.2 2123.20  4717.5 2118.08  4745.8 2115.47  4759.9 2115.95  4788.2 2115.20
  4802.4 2113.46  4816.5 2112.87  4844.8 2107.43  4901.4 2105.09  4929.6 2099.74
  4932.2 2095.34  4936.2 2093.34  4979.6 2093.34  4983.6 2095.34  4986.2 2099.67
  5002.9 2098.88  5030.4 2105.64  5050.4 2106.70  5070.4 2105.77  5140.4 2106.13
  5220.4 2113.10  5240.4 2112.00  5310.4 2116.66  5400.4 2116.77  5531.6 2114.71
#Mann=3,-1,0
  4434.7    0.05       0  4932.2    0.05       0  4983.6    0.05       0
Bank Sta=4932.2,4983.6
Exp/Cntr=0.3,0.1

Type RM Length L Ch R = 1,1056090,940,940,940
BEGIN DESCRIPTION:
Clear Fork Brazos Rv 328.0
END DESCRIPTION:
XS GIS Cut Line= 3
      1309190.82      6950784.03      1309807.48      6950043.45
      1309866.42      6949682.03
#Sta/Elev= 30
  4036.3 2114.35  4221.2 2114.42  4348.8 2112.43  4398.2 2110.06  4447.7 2112.63
  4469.8 2111.16  4490.7 2112.13  4540.1 2108.75  4626.0 2108.16  4682.0 2105.71
  4767.9 2106.77  4817.4 2103.94  4959.3 2102.96  4973.6 2101.89  4987.9 2098.89
  4994.2 2099.18  4996.3 2093.29  4998.3 2091.29  5020.0 2091.29  5022.0 2093.29
  5025.8 2097.97  5046.1 2104.57  5157.5 2102.49  5238.6 2102.88  5299.4 2106.63
  5319.6 2108.62  5325.5 2110.63  5330.6 2109.62  5339.9 2111.41  5366.2 2111.89
#Mann=3,-1,0
  4036.3    0.05       0  4996.3    0.05       0  5022.0    0.05       0
Bank Sta=4996.3,5022
Exp/Cntr=0.3,0.1

Type RM Length L Ch R = 1,1055150,387,387,387
BEGIN DESCRIPTION:
Mapping XS d27c41ea
END DESCRIPTION:
XS GIS Cut Line= 3
      1309496.39      6951485.41      1309968.60      6951138.19
      1310121.25      6950132.13
#Sta/Elev= 30
  4094.4 2115.07  4192.0 2113.99  4241.6 2114.53  4263.8 2113.76  4449.7 2113.51
  4761.6 2110.36  4923.5 2110.17  4957.7 2109.26  4963.9 2107.88  4984.1 2101.59
  4989.3 2093.64  4991.3 2091.64  5013.1 2091.64  5015.1 2093.64  5021.4 2099.17
  5026.4 2098.60  5034.7 2100.32  5055.0 2101.73  5115.6 2102.18  5135.9 2103.66
  5158.8 2103.99  5196.6 2102.72  5227.5 2102.69  5257.2 2106.48  5286.2 2109.15
  5348.3 2108.69  5429.2 2112.46  5624.8 2111.50  5661.8 2112.35  5698.1 2111.68
#Mann=3,-1,0
  4094.4    0.05       0  4989.3    0.05       0  5015.1    0.05       0
Bank Sta=4989.3,5015.1
Exp/Cntr=0.3,0.1

Type RM Length L Ch R = 1,1054763,413,413,413
BEGIN DESCRIPTION:
Clear Fork Brazos Rv 327.0
END DESCRIPTION:
XS GIS Cut Line= 3
      1310628.31      6951624.27      1310378.32      6950742.36
      1310225.55      6950124.32
#Sta/Elev= 30
  4059.0 2119.95  4252.6 2114.99  4567.9 2112.01  4658.0 2106.05  4793.1 2100.51
  4821.0 2100.54  4845.1 2098.54  4854.9 2098.77  4865.9 2104.33  4876.2 2104.47
  4894.0 2100.97  4949.0 2102.44  4972.3 2101.40  4975.3 2096.56  4980.5 2096.56
  4982.4 2093.12  4984.4 2091.12  5006.1 2091.12  5008.1 2093.12  5021.4 2101.10
  5031.7 2100.85  5042.0 2102.42  5072.9 2103.05  5173.9 2101.41  5215.3 2106.60
  5220.5 2105.83  5256.8 2109.62  5261.9 2109.11  5298.2 2111.48  5612.3 2111.17
#Mann=3,-1,0
  4059.0    0.05       0  4982.4    0.05       0  5008.1    0.05       0
Bank Sta=4982.4,5008.1
Exp/Cntr=0.3,0.1

Type RM Length L Ch R = 1,1054350,543,543,543
BEGIN DESCRIPTION:
Clear Fork Brazos Rv 326.0
END DESCRIPTION:
XS GIS Cut Line= 3
      1310989.44      6951659.03      1310705.00      6950488.00
      1310579.85      6950034.53
#Sta/Elev= 30
  3800.6 2129.04  3863.4 2127.20  3880.9 2125.79  3964.4 2122.37  4089.7 2119.43
  4136.6 2117.41  4183.5 2116.34  4367.6 2113.74  4601.2 2112.71  4655.8 2110.23
  4684.7 2109.92  4768.2 2102.43  4830.7 2100.70  4903.8 2100.70  4945.6 2099.33
  4964.5 2097.38  4984.7 2091.84  4986.7 2089.84  5008.7 2089.84  5010.7 2091.84
  5016.0 2096.96  5022.9 2102.28  5028.0 2101.79  5036.8 2107.72  5047.2 2108.38
  5057.2 2110.27  5175.8 2109.93  5182.0 2110.67  5210.2 2109.61  5476.1 2109.10
#Mann=3,-1,0
  3800.6    0.05       0  4984.7    0.05       0  5010.7    0.05       0
Bank Sta=4984.7,5010.7
Exp/Cntr=0.3,0.1

Type RM Length L Ch R = 1,1053807,537,537,537
BEGIN DESCRIPTION:
Clear Fork Brazos Rv 325.0
END DESCRIPTION:
XS GIS Cut Line= 4
      1311084.97      6951234.26      1311268.27      6950666.06
      1311205.00      6950438.00      1310920.02      6949985.47
#Sta/Elev= 30
  4164.9 2115.44  4312.5 2110.53  4344.5 2109.17  4376.5 2106.18  4477.9 2102.93
  4542.0 2107.93  4670.2 2107.60  4675.8 2108.88  4686.3 2107.54  4828.8 2106.06
  4884.5 2107.83  4902.6 2107.13  4926.0 2101.60  4947.2 2098.85  4967.5 2099.50
  4976.3 2097.41  4981.5 2094.32  4985.1 2088.42  4987.1 2086.42  5009.0 2086.42
  5011.0 2088.42  5012.2 2095.56  5021.5 2099.51  5027.5 2100.02  5158.1 2099.98
  5173.4 2100.61  5200.5 2104.43  5231.1 2104.24  5340.6 2108.25  5533.4 2107.45
#Mann=3,-1,0
  4164.9    0.05       0  4985.1    0.03       0  5011.0    0.05       0
Bank Sta=4985.1,5011
Exp/Cntr=0.3,0.1

Type RM Length L Ch R = 1,1053270,934,934,934
BEGIN DESCRIPTION:
Clear Fork Brazos Rv 324.0
END DESCRIPTION:
XS GIS Cut Line= 4
      1311536.35      6951359.04      1311557.21      6950354.44
      1311505.00      6950038.00      1311420.01      6949673.00
#Sta/Elev= 30
  3679.0 2114.41  3790.1 2108.78  3830.1 2108.02  3850.0 2106.08  3855.0 2106.79
  3930.1 2100.77  4070.1 2095.24  4100.1 2096.33  4260.2 2093.61  4460.2 2093.30
  4530.2 2097.44  4550.2 2096.90  4620.2 2101.19  4700.5 2102.53  4872.8 2099.62
  4903.2 2100.14  4964.0 2098.25  4984.3 2096.18  5007.1 2095.75  5009.4 2088.46
  5013.4 2086.46  5057.3 2086.46  5061.3 2088.46  5065.8 2098.07  5076.4 2101.85
  5086.7 2103.05  5113.6 2110.17  5161.3 2110.57  5302.3 2107.27  5379.3 2107.18
#Mann=3,-1,0
  3679.0    0.05       0  5009.4    0.03       0  5061.3    0.05       0
#XS Ineff=2,0
    0.00 4687.50 2104.81 5312.50    0.00 2104.81
Permanent Ineff=
       F       F
Bank Sta=5009.4,5061.3
Exp/Cntr=0.3,0.1

Type RM Length L Ch R = 1,1052336,917,917,917
BEGIN DESCRIPTION:
Clear Fork Brazos Rv 323.0
END DESCRIPTION:
XS GIS Cut Line= 3
      1312065.82      6951152.10      1312086.66      6950610.42
      1312066.40      6950126.12
#Sta/Elev= 30
  4435.1 2125.44  4539.0 2120.69  4599.3 2120.68  4649.4 2114.05  4669.4 2113.18
  4689.4 2108.72  4729.4 2103.98  4779.5 2100.78  4799.2 2098.26  4819.5 2101.08
  4839.5 2098.18  4889.5 2100.15  4919.6 2096.52  4939.6 2096.14  4949.6 2096.08
  4969.6 2098.43  4989.6 2098.17  4996.8 2088.52  4998.8 2086.52  5020.8 2086.52
  5022.8 2088.52  5029.6 2088.00  5049.7 2096.51  5059.7 2097.87  5119.7 2099.10
  5169.8 2097.86  5249.8 2098.67  5289.9 2097.68  5349.9 2103.88  5461.9 2103.87
#Mann=3,-1,0
  4435.1    0.05       0  4996.8    0.05       0  5022.8    0.05       0
Bank Sta=4996.8,5022.8
Exp/Cntr=0.3,0.1

Type RM Length L Ch R = 1,1051419,899,899,899
BEGIN DESCRIPTION:
Clear Fork Brazos Rv 322.0
END DESCRIPTION:
XS GIS Cut Line= 3
      1312447.76      6951492.39      1312860.94      6950190.27
      1312828.87      6949901.85
#Sta/Elev= 30
  3633.9 2113.33  3868.4 2108.05  3911.3 2105.88  3970.5 2104.68  4008.0 2102.09
  4239.1 2099.94  4341.4 2099.78  4414.9 2100.85  4551.3 2100.57  4561.7 2100.00
  4567.0 2098.59  4604.5 2094.70  4719.1 2095.63  4782.1 2094.86  4830.4 2096.73
  4835.7 2096.06  4949.9 2096.52  4964.7 2096.06  4987.0 2084.73  4989.0 2082.73
  5011.0 2082.73  5013.0 2084.73  5022.4 2095.65  5032.5 2096.22  5072.7 2095.47
  5143.1 2091.79  5153.2 2092.79  5173.3 2098.23  5189.0 2099.59  5290.2 2099.60
#Mann=3,-1,0
  3633.9    0.05       0  4987.0    0.05       0  5013.0    0.05       0
#XS Ineff=2,0
    0.00 4709.00 2106.08 5291.00    0.00 2106.08
Permanent Ineff=
       F       F
Bank Sta=4987,5013
Exp/Cntr=0.3,0.1

Type RM Length L Ch R = 1,1050520,1110,1110,1110
BEGIN DESCRIPTION:
Clear Fork Brazos Rv 321.0
END DESCRIPTION:
XS GIS Cut Line= 3
      1312676.94      6951603.46      1313705.00      6950188.00
      1314054.99      6948588.04
#Sta/Elev= 30
  3251.7 2105.53  3532.9 2099.75  4721.7 2096.74  4865.2 2092.35  4943.5 2093.29
  4951.7 2090.98  4958.2 2085.92  4964.4 2088.07  4972.9 2084.30  4980.3 2084.91
  4982.3 2082.91  5005.3 2082.91  5007.3 2084.91  5020.5 2092.52  5025.6 2091.02
  5031.8 2094.19  5328.7 2090.02  5359.4 2093.45  5379.9 2090.33  5410.6 2090.87
  5431.0 2087.28  5446.0 2087.26  5461.8 2090.83  5523.2 2089.85  5538.9 2087.59
  5625.5 2098.79  6168.1 2105.32  6362.6 2114.58  6526.7 2129.05  6638.9 2134.64
#Mann=3,-1,0
  3251.7    0.05       0  4980.3    0.05       0  5007.3    0.05       0
#XS Ineff=2,0
       0                 5330.70    0.00 2105.23
Permanent Ineff=
       F       F
Bank Sta=4980.3,5007.3
Exp/Cntr=0.3,0.1

Type RM Length L Ch R = 1,1049410,551,551,551
BEGIN DESCRIPTION:
Clear Fork Brazos Rv 320.0
END DESCRIPTION:
XS GIS Cut Line= 3
      1312554.99      6952288.01      1314155.00      6950888.00
      1314755.00      6948687.99
#Sta/Elev= 30
  2874.2 2124.49  3058.8 2114.94  3469.8 2101.19  4482.5 2095.95  4653.3 2088.33
  4787.6 2088.45  4880.2 2093.05  4943.8 2089.49  4993.1 2090.92  4996.9 2087.72
  4997.8 2082.79  4999.8 2080.79  5024.9 2082.79  5062.4 2091.12  5155.7 2088.90
  5217.9 2091.93  5694.7 2095.23  6432.0 2096.14  6532.7 2097.53  6693.2 2100.77
  6847.0 2109.10  6907.4 2115.26  6955.8 2125.12  7035.3 2129.29  7052.6 2136.96
  7094.0 2130.64  7135.5 2133.00  7149.3 2136.86  7176.9 2131.75  7280.6 2137.00
#Mann=5,-1,0
  2874.2    0.05       0  4997.8    0.05       0  5024.9    0.05       0
  6432.0    0.12       0  6532.7    0.05       0
#XS Ineff=2,0
    0.00 4834.30 2101.29               0
Permanent Ineff=
       F       F
Bank Sta=4997.8,5024.9
Exp/Cntr=0.3,0.1

Type RM Length L Ch R = 1,1048859,1636,1636,1636
BEGIN DESCRIPTION:
Clear Fork Brazos Rv 319.0
END DESCRIPTION:
XS GIS Cut Line= 3
      1314655.00      6951538.00      1314605.00      6951138.00
      1314805.00      6948738.03
#Sta/Elev= 30
  4594.3 2109.41  4896.6 2102.28  4959.6 2090.26  4967.2 2084.20  4980.1 2082.37
  4982.1 2080.37  5005.2 2080.37  5007.2 2082.37  5007.4 2085.14  5017.5 2089.41
  5027.5 2090.27  5147.9 2086.52  5208.1 2089.47  5416.4 2085.11  5719.9 2084.76
  5777.6 2087.48  5830.3 2085.35  5890.5 2092.79  5950.7 2093.84  6502.3 2093.60
  6628.6 2095.04  6813.7 2100.43  6974.2 2109.05  6986.8 2106.41  6994.3 2109.06
  7134.8 2116.19  7164.9 2121.00  7205.0 2119.79  7325.5 2131.18  7405.7 2135.07
#Mann=5,-1,0
  4594.3    0.05       0  4980.1    0.05       0  5007.2    0.05       0
  6502.3    0.12       0  6628.6    0.05       0
#XS Ineff=2,0
       0                 5471.70    0.00 2106.29
Permanent Ineff=
       F       F
Bank Sta=4980.1,5007.2
Exp/Cntr=0.3,0.1

Type RM Length L Ch R = 1,1047223,243,243,243
BEGIN DESCRIPTION:
Clear Fork Brazos Rv 318.0
END DESCRIPTION:
XS GIS Cut Line= 3
      1314705.00      6951638.00      1315405.00      6950388.00
      1315470.58      6950010.91
#Sta/Elev= 30
  3568.0 2110.10  3641.1 2108.66  3662.8 2109.74  3934.8 2103.48  4133.1 2094.83
  4347.4 2091.29  4397.9 2089.03  4404.7 2086.70  4413.9 2087.82  4419.6 2086.29
  4441.3 2085.77  4516.6 2086.31  4581.7 2084.13  4749.5 2085.80  4759.8 2085.66
  4765.5 2083.34  4794.3 2085.05  4977.7 2086.37  4992.7 2085.94  4997.5 2079.73
  4999.1 2077.73  5017.6 2077.73  5019.2 2079.73  5020.9 2078.23  5027.9 2084.30
  5041.2 2085.86  5102.2 2083.86  5112.3 2084.58  5142.1 2091.43  5383.4 2090.95
#Mann=3,-1,0
  3568.0    0.05       0  4997.5    0.05       0  5019.2    0.05       0
Bank Sta=4997.5,5019.2
Exp/Cntr=0.3,0.1

Type RM Length L Ch R = 1,1046980,1403,1403,1403
BEGIN DESCRIPTION:
Mapping XS 3e9c2f5c
END DESCRIPTION:
XS GIS Cut Line= 3
      1314745.79      6951645.49      1315348.76      6950626.05
      1315764.59      6950422.70
#Sta/Elev= 30
  3521.6 2108.95  3600.0 2109.10  3634.9 2107.11  3681.3 2107.39  3878.2 2102.88
  4006.9 2096.19  4176.6 2091.00  4198.0 2088.66  4204.2 2090.11  4235.1 2091.21
  4299.4 2091.07  4330.7 2089.14  4366.8 2084.50  4650.5 2085.41  4666.1 2084.91
  4671.9 2083.48  4687.6 2083.81  4693.4 2085.05  4867.8 2084.35  4980.1 2085.55
  4991.5 2081.00  4992.5 2078.39  4994.1 2076.39  5012.6 2076.39  5014.2 2078.39
  5030.9 2082.35  5053.4 2084.11  5081.5 2084.00  5098.5 2089.55  5168.9 2090.71
#Mann=3,-1,0
  3521.6    0.05       0  4992.5    0.05       0  5014.2    0.05       0
Bank Sta=4992.5,5014.2
Exp/Cntr=0.3,0.1

Type RM Length L Ch R = 1,1045577,535,535,535
BEGIN DESCRIPTION:
Clear Fork Brazos Rv 317.0
END DESCRIPTION:
XS GIS Cut Line= 3
      1315154.99      6951788.01      1315505.00      6951588.00
      1315873.23      6951294.20
#Sta/Elev= 30
  4596.2 2106.16  4631.5 2104.14  4647.3 2104.04  4749.5 2099.54  4787.0 2098.51
  4792.7 2097.58  4824.4 2096.60  4846.0 2095.11  4851.8 2092.87  4861.1 2090.58
  4889.2 2086.29  4910.8 2084.07  4932.4 2082.25  4954.0 2081.43  4976.3 2082.45
  4985.6 2080.61  4991.4 2078.10  4991.8 2075.74  4993.4 2073.74  5011.9 2073.74
  5013.5 2075.74  5020.9 2081.81  5134.6 2080.77  5184.3 2081.24  5198.7 2082.38
  5205.1 2083.65  5213.1 2083.67  5241.9 2088.42  5411.6 2088.70  5470.4 2087.93
#Mann=3,-1,0
  4596.2    0.05       0  4991.8    0.05       0  5013.5    0.05       0
Bank Sta=4991.8,5013.5
Exp/Cntr=0.3,0.1

Type RM Length L Ch R = 1,1045042,478,478,478
BEGIN DESCRIPTION:
Clear Fork Brazos Rv 316.0
END DESCRIPTION:
XS GIS Cut Line= 3
      1315537.23      6952303.30      1315955.00      6951838.00
      1316122.92      6951614.10
#Sta/Elev= 30
  4381.2 2102.65  4461.2 2098.50  4489.6 2098.68  4510.5 2095.49  4546.4 2094.94
  4581.6 2092.14  4616.8 2092.24  4645.1 2090.11  4666.8 2090.32  4695.2 2089.35
  4701.9 2088.24  4744.5 2088.09  4779.6 2085.13  4787.1 2086.25  4793.9 2084.99
  4801.3 2086.16  4815.5 2085.61  4850.7 2079.54  4921.7 2081.32  4956.8 2080.93
  4975.5 2072.36  4977.5 2070.36  5000.7 2070.36  5002.7 2072.36  5003.2 2081.25
  5049.2 2078.90  5084.7 2083.55  5149.2 2083.93  5213.8 2086.91  5286.4 2086.75
#Mann=3,-1,0
  4381.2    0.05       0  4975.5    0.05       0  5002.7    0.05       0
Bank Sta=4975.5,5002.7
Exp/Cntr=0.3,0.1

Type RM Length L Ch R = 1,1044564,1063,1063,1063
BEGIN DESCRIPTION:
Clear Fork Brazos Rv 315.0
END DESCRIPTION:
XS GIS Cut Line= 5
      1315704.97      6952388.01      1316259.83      6952198.01
      1316619.55      6951830.06      1316662.24      6951528.98
      1316533.76      6950966.43
#Sta/Elev= 30
  4422.0 2098.36  4443.2 2095.69  4526.3 2089.40  4562.8 2089.33  4601.7 2087.07
  4770.8 2085.07  4807.9 2084.96  4813.2 2085.84  4876.5 2084.46  4918.8 2085.04
  4933.0 2084.13  4964.3 2077.57  4971.7 2080.06  4990.3 2079.98  4991.5 2071.83
  4993.5 2069.83  5016.7 2069.83  5018.7 2071.83  5019.3 2073.25  5033.4 2080.11
  5040.4 2080.74  5203.2 2078.89  5330.3 2079.70  5478.9 2078.13  5565.5 2084.37
  5626.1 2083.79  5656.4 2082.20  5717.1 2082.11  5992.3 2085.42  6404.2 2086.59
#Mann=3,-1,0
  4422.0    0.05       0  4991.5    0.05       0  5018.7    0.05       0
Bank Sta=4991.5,5018.7
Exp/Cntr=0.3,0.1

Type RM Length L Ch R = 1,1043501,1264,1264,1264
BEGIN DESCRIPTION:
Clear Fork Brazos Rv 314.0
END DESCRIPTION:
XS GIS Cut Line= 3
      1315692.09      6952921.98      1317218.17      6952432.39
      1318150.24      6951937.71
#Sta/Elev= 30
  3376.1 2085.43  3405.5 2085.91  3431.7 2084.81  3699.8 2083.02  3872.8 2083.25
  4090.5 2081.89  4513.3 2081.67  4639.4 2082.55  4684.4 2081.96  4743.4 2077.17
  4954.5 2077.96  4965.0 2075.91  4977.8 2069.25  4986.5 2070.97  4995.5 2075.71
  5001.2 2076.37  5004.2 2070.57  5006.2 2068.57  5029.4 2068.57  5031.4 2070.57
  5031.8 2076.91  5099.7 2080.99  5336.0 2080.01  5348.8 2080.69  5379.9 2079.97
  5621.8 2080.42  5726.1 2081.97  5852.3 2082.36  5978.6 2087.16  6034.0 2087.42
#Mann=3,-1,0
  3376.1    0.05       0  5004.2    0.05       0  5031.4    0.05       0
Bank Sta=5004.2,5031.4
Exp/Cntr=0.3,0.1

Type RM Length L Ch R = 1,1042237,1126,1126,1126
BEGIN DESCRIPTION:
Clear Fork Brazos Rv 313.0
END DESCRIPTION:
XS GIS Cut Line= 3
      1316005.04      6954387.97      1317605.00      6953438.00
      1318119.22      6952322.99
#Sta/Elev= 30
  3132.0 2095.63  3336.5 2087.24  3373.6 2087.32  3416.4 2084.41  3656.1 2079.75
  4504.3 2076.57  4883.6 2079.50  4899.2 2078.19  4911.3 2074.72  4963.5 2075.18
  4981.0 2067.68  4983.0 2065.68  5006.7 2065.68  5008.7 2067.68  5014.8 2072.65
  5036.8 2075.13  5144.7 2074.18  5173.1 2072.25  5196.1 2074.39  5247.5 2074.42
  5316.3 2078.89  5444.2 2074.77  5488.3 2077.28  5686.5 2078.06  5752.6 2081.21
  5807.6 2081.04  5950.8 2085.99  5981.0 2085.31  6032.4 2088.60  6220.6 2090.16
#Mann=3,-1,0
  3132.0    0.05       0  4981.0    0.05       0  5008.7    0.05       0
Bank Sta=4981,5008.7
Exp/Cntr=0.3,0.1

Type RM Length L Ch R = 1,1041111,554,554,554
BEGIN DESCRIPTION:
Clear Fork Brazos Rv 312.0
END DESCRIPTION:
XS GIS Cut Line= 3
      1316506.77      6954946.38      1318505.00      6953288.00
      1318255.00      6951687.97
#Sta/Elev= 30
  2413.0 2091.04  2488.7 2090.09  2602.7 2084.90  2773.3 2080.41  2878.7 2080.99
  3085.8 2076.88  3291.5 2075.41  3682.2 2076.94  4669.2 2077.47  4811.2 2072.15
  4959.6 2072.41  4988.3 2069.23  4989.4 2065.64  4991.4 2063.64  5015.2 2063.64
  5017.2 2065.64  5038.6 2072.62  5060.4 2074.13  5080.6 2077.48  5151.5 2080.68
  5181.8 2079.59  5212.2 2080.76  5435.4 2080.55  5708.1 2083.63  5822.0 2082.76
  5947.5 2083.75  6042.1 2086.37  6285.0 2086.38  6568.4 2091.32  6629.2 2091.13
#Mann=3,-1,0
  2413.0    0.05       0  4989.4    0.05       0  5017.2    0.05       0
Bank Sta=4989.4,5017.2
Exp/Cntr=0.3,0.1

Type RM Length L Ch R = 1,1040557,542,542,542
BEGIN DESCRIPTION:
Clear Fork Brazos Rv 311.0
END DESCRIPTION:
XS GIS Cut Line= 3
      1316576.27      6955093.91      1318705.00      6953788.00
      1319705.01      6951387.98
#Sta/Elev= 30
  2498.9 2090.28  2560.0 2089.92  2691.4 2083.25  2859.6 2078.06  3097.5 2077.85
  3295.2 2075.03  4093.3 2073.99  4240.2 2075.56  4872.5 2075.04  4946.0 2070.14
  4982.7 2071.08  4982.8 2064.64  4984.8 2062.64  5008.6 2062.64  5010.6 2064.64
  5010.9 2069.32  5017.9 2071.69  5147.9 2070.72  5194.0 2075.92  5820.1 2073.79
  6494.0 2076.72  6577.9 2078.45  6618.6 2077.27  7108.8 2081.22  7292.4 2084.46
  7398.6 2088.48  7422.4 2087.28  7534.0 2089.23  7581.6 2092.25  7596.3 2091.21
#Mann=3,-1,0
  2498.9    0.05       0  4982.8    0.03       0  5010.6    0.05       0
Bank Sta=4982.8,5010.6
Exp/Cntr=0.3,0.1

Type RM Length L Ch R = 1,1040015,1668,1668,1668
BEGIN DESCRIPTION:
Clear Fork Brazos Rv 310.0
END DESCRIPTION:
XS GIS Cut Line= 3
      1317782.82      6955363.04      1319005.00      6954188.00
      1320004.99      6950988.03
#Sta/Elev= 30
  3304.7 2074.34  3338.0 2071.78  3776.7 2071.13  4908.1 2073.17  4978.9 2070.01
  4982.7 2065.06  4984.7 2063.06  5008.4 2063.06  5010.4 2065.06  5021.6 2070.57
  5031.5 2071.16  5241.1 2068.49  5440.1 2074.59  6079.2 2073.15  6195.0 2070.37
  6324.9 2070.91  6362.6 2073.72  6627.7 2072.89  6770.7 2075.71  6865.5 2073.36
  6995.4 2077.19  7260.5 2079.48  7650.8 2087.98  7776.5 2088.67  7833.6 2091.87
  7891.7 2091.74  7944.1 2095.00  8059.4 2097.33  8168.9 2103.71  8352.7 2108.64
#Mann=3,-1,0
  3304.7    0.05       0  4982.7    0.05       0  5010.4    0.05       0
#XS Ineff=2,0
       0                 5454.50    0.00 2075.87
Permanent Ineff=
       F       F
Bank Sta=4982.7,5010.4
Exp/Cntr=0.3,0.1

Type RM Length L Ch R = 1,1038347,1402,1402,1402
BEGIN DESCRIPTION:
Clear Fork Brazos Rv 309.0
END DESCRIPTION:
XS GIS Cut Line= 3
      1318609.31      6955454.85      1319955.00      6954188.00
      1320172.57      6951653.90
#Sta/Elev= 30
  3150.9 2072.92  3181.0 2070.14  3739.8 2070.68  3803.7 2072.92  3930.7 2071.30
  4334.1 2071.70  4383.5 2069.30  4433.3 2071.48  4786.9 2074.13  4854.8 2072.75
  4892.9 2065.96  4962.6 2066.37  4971.0 2064.62  4975.1 2061.75  4977.1 2059.75
  5000.8 2059.75  5002.8 2061.75  5009.1 2066.89  5060.9 2065.62  5119.5 2070.91
  5256.5 2073.70  5400.6 2072.59  5516.9 2069.32  5568.7 2070.66  5615.0 2071.48
  5622.7 2071.52  6906.1 2078.69  7036.6 2080.51  7297.5 2089.29  7542.5 2094.36
#Mann=9,-1,0
  3150.9    0.05       0  4854.8    0.12       0  4975.1    0.07       0
  5002.8    0.12       0  5256.5    0.05       0  5516.9    0.12       0
  5568.7    0.05       0  5615.0    0.12       0  5622.7    0.05       0
#XS Ineff=2,0
       0                 5271.00    0.00 2074.98
Permanent Ineff=
       F       F
Bank Sta=4975.1,5002.8
Exp/Cntr=0.3,0.1

Type RM Length L Ch R = 1,1036945,586,586,586
BEGIN DESCRIPTION:
Clear Fork Brazos Rv 308.0
END DESCRIPTION:
XS GIS Cut Line= 4
      1319362.35      6955540.29      1319620.93      6955137.59
      1320805.00      6954638.00      1323277.46      6953539.34
#Sta/Elev= 30
  3236.6 2071.74  3275.1 2068.06  3347.8 2070.12  3826.3 2071.05  4360.0 2069.46
  4739.8 2070.94  4803.5 2067.21  4880.0 2067.74  4938.3 2063.10  4978.6 2063.81
  4984.8 2055.79  4986.8 2053.79  5010.9 2053.79  5012.9 2055.79  5014.7 2058.83
  5022.2 2064.14  5066.7 2062.44  5153.5 2069.07  5206.2 2060.40  5267.8 2061.53
  5281.4 2063.27  5333.4 2062.69  5379.9 2067.96  5455.2 2070.66  5766.3 2074.99
  5918.9 2079.52  6083.7 2081.28  6787.6 2081.80  7199.4 2087.73  7705.9 2091.77
#Mann=4,-1,0
  3236.6    0.05       0  4984.8    0.07       0  5012.9    0.05       0
  5267.8    0.05       0
#XS Ineff=2,0
       0                 5155.30    0.00 2070.40
Permanent Ineff=
       F       F
Bank Sta=4984.8,5012.9
Exp/Cntr=0.3,0.1

Type RM Length L Ch R = 1,1036359,1108,1108,1108
BEGIN DESCRIPTION:
Mapping XS 7fa8f23c
END DESCRIPTION:
XS GIS Cut Line= 3
      1319989.26      6955600.38      1320543.26      6955371.70
      1322027.15      6954642.77
#Sta/Elev= 30
  3954.9 2070.51  4023.6 2066.68  4029.0 2068.13  4076.9 2068.70  4668.9 2068.08
  4843.2 2070.34  4879.3 2069.63  4894.4 2066.64  4923.8 2062.86  4933.1 2063.74
  4955.6 2062.56  4961.2 2057.78  4975.0 2054.82  4977.0 2052.82  5001.2 2052.82
  5003.2 2054.82  5006.2 2062.74  5045.5 2060.10  5078.5 2061.84  5157.8 2063.18
  5253.5 2071.25  5380.6 2070.50  5478.3 2071.84  5483.8 2070.24  5500.8 2072.59
  5506.3 2069.92  5514.3 2072.88  5737.2 2081.66  6060.3 2085.02  6207.5 2084.93
#Mann=5,-1,0
  3954.9    0.05       0  4894.4    0.12       0  4975.0    0.07       0
  5003.2    0.12       0  5078.5    0.05       0
Bank Sta=4975,5003.2
Exp/Cntr=0.3,0.1

Type RM Length L Ch R = 1,1035251,336,336,336
BEGIN DESCRIPTION:
Mapping XS 8b60b616
END DESCRIPTION:
XS GIS Cut Line= 3
      1320300.86      6955536.56      1321372.79      6955627.32
      1322207.56      6955700.07
#Sta/Elev= 30
  3490.1 2068.20  3825.4 2068.35  3965.9 2067.70  4155.3 2068.58  4337.3 2068.05
  4407.5 2068.52  4698.6 2067.84  4788.9 2063.91  4869.2 2063.51  4929.4 2064.01
  4959.6 2060.15  4969.6 2060.12  4999.7 2058.18  5000.7 2052.98  5002.7 2050.98
  5027.1 2050.98  5029.1 2052.98  5029.8 2051.48  5039.9 2056.65  5049.9 2059.96
  5100.1 2059.41  5110.1 2058.75  5140.2 2061.59  5160.3 2068.32  5180.4 2073.04
  5190.4 2071.13  5200.5 2070.80  5211.3 2072.43  5324.1 2071.18  5403.8 2071.28
#Mann=3,-1,0
  3490.1    0.05       0  5000.7    0.03       0  5029.1    0.05       0
Bank Sta=5000.7,5029.1
Exp/Cntr=0.3,0.1

Type RM Length L Ch R = 1,1034915,815,815,815
BEGIN DESCRIPTION:
Mapping XS bcda02c0
END DESCRIPTION:
XS GIS Cut Line= 2
      1320064.42      6955845.98      1322170.11      6956009.10
#Sta/Elev= 30
  3209.6 2067.81  3330.5 2068.30  3340.6 2067.55  3481.0 2067.04  3511.1 2067.63
  3551.2 2066.39  3641.5 2065.93  3852.1 2066.02  4202.5 2067.57  4744.8 2066.98
  4815.0 2065.38  4825.0 2064.52  4845.1 2060.19  4875.2 2058.50  4885.2 2059.08
  4915.3 2058.22  4965.4 2058.93  4973.6 2052.90  4975.6 2050.90  5000.0 2050.90
  5002.0 2052.90  5005.5 2058.26  5015.6 2058.99  5025.6 2061.93  5035.6 2063.44
  5045.7 2063.51  5095.8 2067.52  5117.0 2066.73  5206.1 2066.12  5321.6 2066.16
#Mann=3,-1,0
  3209.6    0.05       0  4973.6    0.05       0  5002.0    0.05       0
Bank Sta=4973.6,5002
Exp/Cntr=0.3,0.1

Type RM Length L Ch R = 1,1034100,1213,1213,1213
BEGIN DESCRIPTION:
Clear Fork Brazos Rv 300.0
END DESCRIPTION:
XS GIS Cut Line= 3
      1321318.82      6957189.36      1322117.47      6956625.10
      1322195.59      6956112.99
#Sta/Elev= 30
  4226.8 2063.04  4518.6 2063.86  4699.6 2062.81  4762.4 2063.71  4834.3 2063.57
  4848.5 2062.73  4871.1 2063.53  4899.0 2063.20  4907.7 2063.02  4920.0 2059.34
  4943.4 2055.94  4964.3 2057.49  4970.4 2056.12  4974.3 2050.90  4976.3 2048.90
  5000.8 2048.90  5002.8 2050.90  5006.1 2057.91  5014.8 2058.12  5136.6 2056.39
  5211.9 2057.20  5252.3 2055.39  5262.4 2055.53  5287.7 2057.88  5302.9 2058.09
  5323.1 2060.18  5363.6 2062.64  5488.4 2061.82  5556.9 2064.44  5722.7 2064.83
#Mann=3,-1,0
  4226.8    0.05       0  4974.3    0.05       0  5002.8    0.05       0
Bank Sta=4974.3,5002.8
Exp/Cntr=0.3,0.1

Type RM Length L Ch R = 1,1032887,555,555,555
BEGIN DESCRIPTION:
Clear Fork Brazos Rv 299.0
END DESCRIPTION:
XS GIS Cut Line= 3
      1321409.55      6957601.21      1322905.00      6957338.00
      1324155.02      6956187.98
#Sta/Elev= 30
  3474.3 2061.81  3691.4 2061.13  3869.3 2062.36  4251.5 2060.50  4282.0 2055.28
  4302.3 2053.78  4328.5 2054.44  4333.6 2057.19  4373.4 2052.60  4424.1 2051.95
  4657.7 2053.90  4999.8 2054.54  4999.9 2048.70  5001.9 2046.70  5026.3 2046.70
  5028.3 2048.70  5042.4 2054.48  5049.2 2054.57  5211.9 2052.74  5261.8 2050.88
  5282.8 2053.60  5304.4 2059.11  5672.2 2060.06  5707.6 2059.06  5714.4 2060.79
  5813.6 2060.91  5969.6 2063.63  6195.9 2070.93  6578.1 2086.93  6691.3 2089.98
#Mann=3,-1,0
  3474.3    0.05       0  4999.9    0.03       0  5028.3    0.05       0
Bank Sta=4999.9,5028.3
Exp/Cntr=0.3,0.1

Type RM Length L Ch R = 1,1032332,819,819,819
BEGIN DESCRIPTION:
Clear Fork Brazos Rv 298.0
END DESCRIPTION:
XS GIS Cut Line= 3
      1321404.97      6958588.01      1323005.00      6957788.00
      1324255.01      6956187.99
#Sta/Elev= 30
  3216.8 2074.62  3700.4 2063.26  4035.8 2060.65  4214.7 2051.08  4320.9 2052.13
  4365.6 2058.42  4401.9 2051.90  4455.1 2051.78  4460.6 2048.27  4513.8 2051.57
  4790.5 2051.62  4840.8 2055.00  4983.3 2052.61  4991.7 2049.69  4992.3 2046.97
  4994.3 2044.97  5020.7 2046.97  5027.4 2051.75  5041.9 2053.32  5126.9 2051.75
  5191.1 2046.63  5197.4 2051.74  5220.0 2053.86  5226.4 2057.67  5240.8 2055.35
  5261.6 2059.41  6109.7 2059.26  6359.6 2065.25  6757.5 2083.41  7036.1 2091.79
#Mann=3,-1,0
  3216.8    0.05       0  4992.3    0.05       0  5020.7    0.05       0
Bank Sta=4992.3,5020.7
Exp/Cntr=0.3,0.1

Type RM Length L Ch R = 1,1031513,603,603,603
BEGIN DESCRIPTION:
Clear Fork Brazos Rv 297.0
END DESCRIPTION:
XS GIS Cut Line= 3
      1321180.76      6958797.90      1323468.52      6958252.36
      1324893.97      6956686.12
#Sta/Elev= 30
  2614.6 2069.98  2999.3 2071.69  3498.0 2062.39  4690.1 2054.65  4757.3 2045.94
  4792.3 2050.12  4866.2 2050.58  4883.5 2050.16  4973.9 2051.38  4981.4 2050.93
  4985.9 2045.20  4987.9 2043.20  5014.5 2043.20  5016.5 2045.20  5023.9 2050.08
  5071.0 2050.21  5405.7 2049.24  5434.1 2052.06  5441.5 2055.84  5455.7 2057.40
  5498.3 2056.92  5505.0 2054.38  5526.6 2057.14  5568.5 2054.84  6333.4 2060.64
  6446.3 2064.92  6460.5 2062.82  6517.2 2064.09  6553.0 2067.27  7084.3 2083.80
#Mann=7,-1,0
  2614.6    0.05       0  4690.1    0.12       0  4866.2    0.05       0
  4883.5    0.12       0  4985.9    0.07       0  5016.5    0.12       0
  5071.0    0.05       0
Bank Sta=4985.9,5016.5
Exp/Cntr=0.3,0.1

Type RM Length L Ch R = 1,1030910,1426,1426,1426
BEGIN DESCRIPTION:
Clear Fork Brazos Rv 296.0
END DESCRIPTION:
XS GIS Cut Line= 3
      1321462.31      6958956.30      1323605.00      6958738.00
      1326425.02      6958357.96
#Sta/Elev= 30
  2846.2 2065.99  3562.6 2059.96  4718.5 2055.61  4753.5 2053.95  4798.9 2046.78
  4914.1 2049.03  4979.9 2049.29  4985.0 2046.48  4989.7 2043.89  4991.7 2041.89
  5018.4 2041.89  5020.4 2043.89  5030.3 2049.39  5060.5 2048.03  5109.1 2054.38
  5192.0 2057.54  5322.9 2053.76  5898.0 2056.10  6140.2 2053.50  6536.8 2053.42
  6609.6 2056.04  6634.6 2054.40  6682.3 2057.61  7038.2 2058.02  7189.6 2060.81
  7279.5 2059.74  7401.5 2063.05  7430.0 2061.82  7580.6 2064.88  7845.5 2066.31
#Mann=5,-1,0
  2846.2    0.05       0  4914.1    0.12       0  4985.0    0.05       0
  4989.7    0.05       0  5020.4    0.05       0
Bank Sta=4989.7,5020.4
Exp/Cntr=0.3,0.1

Type RM Length L Ch R = 1,1029484,1397,1397,1397
BEGIN DESCRIPTION:
Clear Fork Brazos Rv 295.0
END DESCRIPTION:
XS GIS Cut Line= 3
      1321855.04      6959988.00      1323855.00      6959988.00
      1326865.03      6958481.13
#Sta/Elev= 30
  2993.4 2079.55  3383.4 2069.94  3483.4 2070.88  3753.4 2067.83  3863.4 2063.77
  4083.4 2060.17  4493.4 2065.30  4873.4 2051.26  4913.4 2047.08  4996.2 2046.13
  4996.7 2037.72  4998.7 2035.72  5025.4 2035.72  5027.4 2037.72  5038.1 2042.90
  5052.0 2045.37  5255.6 2046.43  5337.0 2047.07  5432.0 2052.78  5485.4 2052.33
  5507.8 2054.25  5521.4 2052.22  6767.6 2050.83  7169.9 2060.33  7421.4 2060.74
  7460.5 2062.69  7722.0 2064.75  7795.8 2068.25  7818.1 2066.24  8359.5 2073.02
#Mann=5,-1,0
  2993.4    0.05       0  4996.7    0.05       0  5027.4    0.05       0
  5255.6    0.12       0  5432.0    0.05       0
Bank Sta=4996.7,5027.4
Exp/Cntr=0.3,0.1
