HEC-RAS study Clear Fork Brazos Rv.prj: Clear Fork Brazos Rv Base Level Engineering

--- Clear Fork Brazos Rv.g01 (geometry) --- (continued)

Type RM Length L Ch R = 1,1028087,1431,1431,1431
BEGIN DESCRIPTION:
Clear Fork Brazos Rv 294.0
END DESCRIPTION:
XS GIS Cut Line= 3
      1321755.04      6960038.01      1324755.00      6960938.00
      1327454.97      6959438.02
#Sta/Elev= 30
  1874.3 2080.20  1890.8 2079.81  1896.0 2076.89  2209.2 2072.82  2418.0 2065.38
  2469.4 2066.39  2907.8 2057.28  3286.3 2057.33  3816.2 2050.24  4703.6 2049.74
  4847.1 2042.74  4912.4 2044.82  4951.5 2037.73  4956.8 2043.56  4972.1 2034.69
  4974.1 2032.69  5000.9 2032.69  5002.9 2034.69  5003.7 2044.18  5109.3 2043.17
  5189.4 2050.51  5212.3 2048.16  5226.0 2050.11  5418.2 2047.46  6683.4 2051.52
  7214.2 2061.94  7301.1 2066.10  7534.5 2067.56  7637.5 2072.35  8095.0 2076.30
#Mann=3,-1,0
  1874.3    0.05       0  4972.1    0.05       0  5002.9    0.05       0
#XS Ineff=2,0
       0                 6325.30    0.00 2063.73
Permanent Ineff=
       F       F
Bank Sta=4972.1,5002.9
Exp/Cntr=0.3,0.1

Type RM Length L Ch R = 1,1026656,727,727,727
BEGIN DESCRIPTION:
Clear Fork Brazos Rv 293.0
END DESCRIPTION:
XS GIS Cut Line= 3
      1324455.02      6962737.96      1324755.00      6962038.00
      1327155.02      6959937.98
#Sta/Elev= 30
  4237.6 2066.48  4756.1 2053.09  4937.5 2053.47  4955.6 2055.85  4966.5 2050.04
  4977.4 2048.84  4984.6 2043.57  4990.1 2038.89  4990.8 2028.59  4992.8 2026.59
  5020.1 2026.59  5022.1 2028.59  5027.1 2037.09  5034.7 2040.47  5061.2 2040.64
  5105.4 2038.46  5169.5 2045.63  6175.6 2044.86  6302.7 2047.09  6359.7 2051.49
  6445.1 2047.02  6543.8 2046.15  7401.8 2048.51  7628.7 2053.34  7678.0 2056.67
  7698.9 2055.71  7827.0 2060.00  8025.4 2068.60  8046.3 2067.59  8188.2 2072.22
#Mann=5,-1,0
  4237.6    0.05       0  4990.8    0.05       0  5022.1    0.05       0
  5061.2    0.12       0  5169.5    0.05       0
#XS Ineff=2,0
       0                 6328.70    0.00 2056.25
Permanent Ineff=
       F       F
Bank Sta=4990.8,5022.1
Exp/Cntr=0.3,0.1

Type RM Length L Ch R = 1,1025929,707,707,707
BEGIN DESCRIPTION:
Clear Fork Brazos Rv 292.0
END DESCRIPTION:
XS GIS Cut Line= 3
      1324654.98      6963188.02      1325355.00      6962388.00
      1327455.02      6959687.97
#Sta/Elev= 30
  3936.8 2079.66  4007.5 2078.08  4085.4 2071.03  4107.2 2071.19  4121.4 2068.42
  4142.3 2068.69  4163.2 2065.43  4234.4 2062.48  4596.0 2058.79  4631.1 2054.30
  4773.7 2046.98  4829.5 2042.52  4907.3 2040.85  4964.2 2032.29  4973.6 2028.03
  4975.6 2026.03  5002.9 2026.03  5004.9 2028.03  5007.1 2034.22  5063.9 2039.24
  5264.1 2038.97  5519.3 2044.21  7202.4 2047.49  7465.7 2052.70  7635.8 2059.62
  7672.9 2059.04  7722.7 2062.64  7892.8 2065.49  8220.4 2076.49  8420.4 2076.99
#Mann=5,-1,0
  3936.8    0.05       0  4773.7     0.1       0  4973.6    0.07       0
  5004.9     0.1       0  5063.9    0.05       0
Bank Sta=4973.6,5004.9
Exp/Cntr=0.3,0.1

Type RM Length L Ch R = 1,1025222,1245,1245,1245
BEGIN DESCRIPTION:
Clear Fork Brazos Rv 291.0
END DESCRIPTION:
XS GIS Cut Line= 3
      1325555.01      6963537.98      1325955.00      6962538.00
      1327455.00      6959838.00
#Sta/Elev= 30
  3926.1 2064.85  3965.1 2061.51  4109.2 2058.59  4378.4 2046.81  4527.9 2044.78
  4572.3 2041.15  4772.9 2043.92  4832.1 2037.70  4934.5 2037.46  4949.3 2033.17
  4970.8 2030.88  4978.5 2027.49  4980.5 2025.49  5007.9 2025.49  5009.9 2027.49
  5011.1 2034.58  5026.0 2037.07  5067.0 2036.76  5106.1 2036.46  5163.3 2043.21
  5222.8 2044.05  5276.5 2041.58  5759.3 2042.22  5943.4 2045.26  6436.5 2044.76
  7062.2 2047.82  7444.3 2056.46  7577.0 2062.75  7753.2 2065.81  8091.8 2076.37
#Mann=4,-1,0
  3926.1    0.05       0  4978.5    0.07       0  5009.9    0.05       0
  5067.0    0.05       0
Bank Sta=4978.5,5009.9
Exp/Cntr=0.3,0.1

Type RM Length L Ch R = 1,1023977,907,907,907
BEGIN DESCRIPTION:
Mapping XS 7f781855
END DESCRIPTION:
XS GIS Cut Line= 3
      1326302.07      6963911.09      1326796.51      6962988.76
      1328108.65      6960915.96
#Sta/Elev= 30
  4290.0 2049.29  4633.9 2041.04  4894.3 2041.67  4916.2 2038.65  4921.9 2040.38
  4960.1 2034.41  4987.5 2021.25  4989.1 2020.25  5012.6 2021.25  5019.7 2029.10
  5031.5 2029.96  5047.8 2035.29  5189.9 2036.48  5217.6 2038.53  5239.5 2042.57
  5277.7 2039.83  5546.6 2037.47  5777.1 2039.10  5807.7 2040.83  5850.0 2039.64
  5965.3 2042.30  6168.7 2040.92  6284.2 2042.47  6698.5 2041.90  6864.1 2044.15
  6900.2 2042.45  7213.0 2043.12  7270.6 2045.34  7610.5 2046.33  7789.7 2050.42
#Mann=3,-1,0
  4290.0    0.05       0  4987.5    0.05       0  5012.6    0.05       0
Bank Sta=4987.5,5012.6
Exp/Cntr=0.3,0.1

Type RM Length L Ch R = 1,1023070,300,300,300
BEGIN DESCRIPTION:
Clear Fork Brazos Rv 288.0
END DESCRIPTION:
XS GIS Cut Line= 3
      1326705.02      6965037.96      1327505.00      6963438.00
      1328405.00      6960438.00
#Sta/Elev= 30
  3211.9 2059.18  3360.0 2057.69  3466.2 2054.16  3538.9 2055.09  3600.4 2052.47
  3896.7 2053.27  4321.5 2045.83  4464.1 2041.22  4911.3 2037.99  4964.4 2033.67
  4978.4 2027.67  4986.7 2028.04  4989.9 2023.48  4991.9 2021.48  5019.3 2021.48
  5021.3 2023.48  5022.5 2026.35  5042.5 2028.87  5050.3 2032.99  5063.4 2033.81
  5220.0 2033.41  5268.7 2036.73  5335.7 2039.01  5950.8 2038.94  7099.2 2042.90
  7652.6 2051.66  7830.0 2059.25  7861.4 2058.53  7924.0 2062.20  8132.8 2067.63
#Mann=3,-1,0
  3211.9    0.05       0  4989.9    0.05       0  5268.7    0.05       0
Bank Sta=4989.9,5021.3
Exp/Cntr=0.3,0.1

Type RM Length L Ch R = 1,1022770,367,367,367
BEGIN DESCRIPTION:
Mapping XS 18e8909a
END DESCRIPTION:
XS GIS Cut Line= 2
      1327445.48      6964992.40      1328104.05      6961991.31
#Sta/Elev= 30
  3556.8 2045.60  3991.3 2048.54  4083.4 2044.19  4114.2 2040.59  4144.9 2033.34
  4165.3 2032.61  4182.6 2033.78  4187.7 2037.87  4267.7 2041.84  4288.2 2041.83
  4308.7 2038.12  4373.1 2038.40  4390.6 2043.60  4411.1 2044.69  4558.6 2037.79
  4574.9 2034.12  4615.8 2030.91  4841.9 2033.86  4963.9 2033.30  4978.4 2029.66
  4984.3 2023.60  4986.3 2021.60  5013.8 2021.60  5015.8 2023.60  5027.3 2026.99
  5045.8 2027.07  5066.0 2032.76  5354.4 2032.69  5404.1 2039.02  6629.3 2041.37
#Mann=3,-1,0
  3556.8    0.05       0  4984.3    0.05       0  5015.8    0.05       0
#XS Ineff=2,0
    0.00 4708.00 2046.98 5250.00    0.00 2046.98
Permanent Ineff=
       F       F
Bank Sta=4984.3,5015.8
Exp/Cntr=0.3,0.1

Type RM Length L Ch R = 1,1022403,866,866,866
BEGIN DESCRIPTION:
Mapping XS c065a330
END DESCRIPTION:
XS GIS Cut Line= 2
      1327637.32      6965743.18      1328496.49      6961847.70
#Sta/Elev= 30
  2884.0 2047.08  3851.9 2036.65  3882.6 2030.90  3903.1 2032.86  3954.3 2029.03
  3985.0 2021.75  4005.5 2022.47  4015.8 2029.60  4036.2 2030.79  4210.3 2026.61
  4323.0 2029.78  4374.2 2025.08  4404.9 2029.84  4497.0 2030.92  4548.2 2036.83
  4565.8 2033.29  4691.6 2030.35  4892.1 2032.57  4984.6 2026.55  4994.3 2022.58
  4996.3 2020.58  5025.8 2022.58  5039.8 2030.88  5050.0 2031.98  5305.9 2033.42
  5326.5 2026.06  5347.0 2033.43  5521.1 2039.94  5686.1 2037.27  6873.1 2042.79
#Mann=3,-1,0
  2884.0    0.05       0  4994.3    0.05       0  5025.8    0.05       0
#XS Ineff=2,0
    0.00 4537.60 2041.36 5244.00    0.00 2041.36
Permanent Ineff=
       F       F
Bank Sta=4994.3,5025.8
Exp/Cntr=0.3,0.1

Type RM Length L Ch R = 1,1021537,1573,1573,1573
BEGIN DESCRIPTION:
Mapping XS 74eb371e
END DESCRIPTION:
XS GIS Cut Line= 3
      1327812.48      6965901.67      1328179.51      6964783.89
      1329614.21      6963174.02
#Sta/Elev= 30
  3114.8 2049.05  3413.4 2040.65  3729.1 2036.21  4038.0 2035.42  4069.9 2034.06
  4096.4 2030.04  4165.3 2028.81  4191.8 2021.83  4202.8 2028.63  4244.9 2029.36
  4512.2 2028.10  4533.1 2022.49  4554.0 2027.60  4589.9 2028.39  4610.8 2031.91
  4809.0 2026.15  4859.1 2028.29  4908.5 2026.68  4965.3 2027.71  4986.2 2026.32
  4993.7 2023.96  4994.3 2020.14  4996.3 2018.14  5023.8 2018.14  5025.8 2020.14
  5049.8 2029.78  5191.9 2033.86  5630.9 2036.85  5694.4 2035.14  6447.7 2036.21
#Mann=3,-1,0
  3114.8    0.05       0  4994.3    0.03       0  5025.8    0.05       0
#XS Ineff=2,0
    0.00 4597.40 2037.87               0
Permanent Ineff=
       F       F
Bank Sta=4994.3,5025.8
Exp/Cntr=0.3,0.1

Type RM Length L Ch R = 1,1019964,1672,1672,1672
BEGIN DESCRIPTION:
Clear Fork Brazos Rv 285.0
END DESCRIPTION:
XS GIS Cut Line= 3
      1327639.35      6966541.21      1329381.59      6964816.57
      1329826.93      6964527.54
#Sta/Elev= 30
  3427.9 2068.34  3625.1 2059.41  3780.7 2056.56  3936.2 2057.01  4183.7 2050.52
  4226.1 2045.60  4565.5 2033.28  4678.7 2033.21  4855.5 2029.11  4897.9 2030.36
  4905.0 2025.79  4926.2 2026.29  4933.3 2023.60  4940.4 2026.15  4954.5 2023.33
  4961.5 2016.74  4972.1 2016.77  4974.1 2014.77  5001.6 2014.77  5003.6 2016.77
  5004.0 2023.69  5018.1 2024.36  5088.8 2025.55  5187.8 2022.56  5428.2 2026.84
  5534.3 2031.94  6053.8 2031.65  6068.9 2033.90  6074.9 2031.68  6410.3 2031.99
#Mann=3,-1,0
  3427.9    0.05       0  4972.1    0.05       0  5003.6    0.05       0
#XS Ineff=2,0
       0                 5505.30    0.00 2043.76
Permanent Ineff=
       F       F
Bank Sta=4972.1,5003.6
Exp/Cntr=0.3,0.1

Type RM Length L Ch R = 1,1018292,728,728,728
BEGIN DESCRIPTION:
Clear Fork Brazos Rv 284.0
END DESCRIPTION:
XS GIS Cut Line= 3
      1327855.04      6966687.98      1329655.00      6965888.00
      1330243.91      6965652.44
#Sta/Elev= 30
  3027.5 2071.25  3186.8 2062.68  3224.4 2062.84  3262.0 2059.58  3383.8 2056.46
  3476.1 2056.76  3519.9 2053.25  3563.7 2053.13  3801.0 2037.08  3974.7 2030.28
  4132.7 2030.67  4171.7 2028.42  4565.7 2026.37  4756.5 2026.22  4791.4 2028.68
  4920.6 2027.40  4936.4 2026.07  4959.6 2009.55  4965.1 2008.70  4966.8 2010.20
  4968.8 2008.20  4996.3 2008.20  4998.3 2010.20  4999.9 2019.73  5104.9 2020.95
  5119.7 2022.06  5144.0 2027.09  5234.2 2025.57  5257.1 2027.24  5631.5 2029.05
#Mann=3,-1,0
  3027.5    0.05       0  4966.8    0.05       0  4998.3    0.05       0
Bank Sta=4966.8,4998.3
Exp/Cntr=0.3,0.1

Type RM Length L Ch R = 1,1017564,1426,1426,1426
BEGIN DESCRIPTION:
Clear Fork Brazos Rv 283.0
END DESCRIPTION:
XS GIS Cut Line= 3
      1328004.95      6966688.00      1330005.00      6966488.00
      1330455.85      6966217.49
#Sta/Elev= 30
  2990.5 2063.46  3161.4 2057.29  3302.1 2056.85  3339.8 2053.60  3392.5 2053.27
  3573.4 2038.35  3724.2 2030.32  3784.5 2030.25  3842.3 2027.47  3975.4 2026.54
  4055.8 2023.92  4477.9 2023.91  4498.0 2022.76  4739.2 2027.03  4809.6 2026.23
  4839.7 2024.96  4859.8 2020.90  4900.0 2016.02  4970.4 2019.45  4990.5 2018.28
  4990.7 2008.67  4992.3 2006.67  5014.3 2006.67  5015.9 2008.67  5035.5 2016.93
  5066.6 2027.20  5082.2 2025.90  5109.4 2028.05  5140.5 2026.36  5526.3 2028.43
#Mann=3,-1,0
  2990.5    0.05       0  4990.7    0.05       0  5015.9    0.05       0
#XS Ineff=2,0
    0.00 4700.00 2037.62               0
Permanent Ineff=
       F       F
Bank Sta=4990.7,5015.9
Exp/Cntr=0.3,0.1

Type RM Length L Ch R = 1,1016138,678,678,678
BEGIN DESCRIPTION:
Clear Fork Brazos Rv 282.0
END DESCRIPTION:
XS GIS Cut Line= 3
      1328079.34      6967561.92      1329905.00      6967438.00
      1330188.37      6967302.63
#Sta/Elev= 30
  3174.9 2054.19  3330.9 2053.08  3381.0 2050.02  3461.2 2049.59  3599.2 2043.19
  3792.0 2039.79  3842.1 2036.59  3872.2 2036.88  3897.3 2034.68  3952.3 2033.95
  3992.4 2030.97  4032.5 2030.78  4112.7 2027.08  4583.8 2022.83  4814.3 2022.03
  4864.4 2024.02  4904.5 2017.91  4984.7 2013.11  4987.0 2005.68  4988.7 2003.68
  5013.1 2003.68  5014.9 2005.68  5018.9 2012.11  5026.9 2015.55  5086.9 2016.88
  5126.7 2024.46  5205.9 2023.93  5259.7 2026.45  5281.8 2023.72  5318.8 2023.57
#Mann=3,-1,0
  3174.9    0.05       0  4987.0    0.05       0  5014.9    0.05       0
Bank Sta=4987,5014.9
Exp/Cntr=0.3,0.1

Type RM Length L Ch R = 1,1015460,670,670,670
BEGIN DESCRIPTION:
Clear Fork Brazos Rv 281.0
END DESCRIPTION:
XS GIS Cut Line= 3
      1328165.33      6968257.53      1329905.00      6968088.00
      1330218.87      6967879.73
#Sta/Elev= 30
  3233.0 2050.00  3443.7 2043.82  3604.4 2040.21  3674.8 2040.07  3735.0 2036.92
  3797.8 2036.93  3845.6 2034.04  4116.8 2030.22  4237.4 2026.69  4297.7 2027.03
  4337.9 2025.24  4589.1 2021.69  4699.6 2021.10  4718.9 2022.31  4790.0 2017.87
  4850.3 2020.78  4932.5 2021.21  4950.8 2020.28  4970.9 2016.36  4978.4 2013.15
  4983.9 2013.15  4990.6 2002.47  4991.9 2000.47  5010.2 2000.47  5011.5 2002.47
  5024.5 2011.30  5081.7 2012.86  5117.7 2021.65  5132.8 2023.42  5357.6 2022.79
#Mann=3,-1,0
  3233.0    0.05       0  4990.6    0.05       0  5011.5    0.05       0
Bank Sta=4990.6,5011.5
Exp/Cntr=0.3,0.1

Type RM Length L Ch R = 1,1014790,711,711,711
BEGIN DESCRIPTION:
Clear Fork Brazos Rv 280.0
END DESCRIPTION:
XS GIS Cut Line= 3
      1328464.86      6969160.06      1330205.00      6968638.00
      1330344.80      6968552.39
#Sta/Elev= 30
  3184.4 2049.04  3204.6 2047.68  3236.8 2043.23  3289.0 2039.10  3309.0 2035.06
  3330.7 2035.34  3347.3 2032.22  3385.5 2033.14  3424.7 2030.38  3445.0 2030.11
  3523.0 2028.89  3581.3 2024.82  3756.7 2024.19  3797.9 2025.50  3803.2 2024.18
  3831.0 2022.91  4406.1 2019.87  4865.4 2019.11  4907.2 2021.38  4969.8 2010.95
  4979.4 2007.34  4983.0 2002.00  4985.0 2000.00  5009.9 2000.00  5011.8 2002.00
  5014.7 2007.58  5024.3 2009.89  5051.5 2012.43  5088.2 2019.42  5165.1 2021.37
#Mann=5,-1,0
  3184.4    0.05       0  3445.0    0.12       0  3756.7    0.05       0
  4983.0    0.05       0  5011.8    0.05       0
Bank Sta=4983,5011.8
Exp/Cntr=0.3,0.1

Type RM Length L Ch R = 1,1014079,706,706,706
BEGIN DESCRIPTION:
Clear Fork Brazos Rv 279.0
END DESCRIPTION:
XS GIS Cut Line= 3
      1328504.98      6970038.01      1330505.00      6969238.00
      1330633.15      6969122.66
#Sta/Elev= 30
  2845.3 2058.59  2943.6 2057.35  3006.9 2054.58  3261.3 2034.58  3491.5 2022.73
  3728.5 2020.27  3912.9 2020.47  3985.6 2019.58  4355.5 2018.78  4654.7 2019.19
  4676.3 2020.16  4718.2 2019.16  4852.6 2018.84  4913.2 2011.49  4936.1 2010.24
  4960.3 2010.36  4977.8 2008.71  4984.6 2006.38  4990.0 2006.95  4990.9 2000.98
  4992.8 1998.98  5017.8 1998.98  5019.7 2000.98  5020.7 2003.38  5027.4 2004.44
  5034.9 2010.25  5055.8 2012.17  5077.5 2017.68  5091.7 2020.20  5171.8 2019.93
#Mann=5,-1,0
  2845.3    0.05       0  4355.5    0.12       0  4718.2    0.05       0
  4990.9    0.05       0  5019.7    0.05       0
Bank Sta=4990.9,5019.7
Exp/Cntr=0.3,0.1

Type RM Length L Ch R = 1,1013373,695,695,695
BEGIN DESCRIPTION:
Clear Fork Brazos Rv 278.0
END DESCRIPTION:
XS GIS Cut Line= 3
      1328704.98      6970288.00      1330705.00      6969888.00
      1331338.04      6969395.64
#Sta/Elev= 30
  2961.6 2054.57  3084.0 2050.23  3145.2 2042.30  3206.4 2042.05  3237.0 2036.33
  3359.3 2028.40  3817.1 2020.95  4004.1 2018.71  4105.7 2018.01  4318.7 2017.16
  4756.5 2019.02  4960.4 2007.92  4980.8 2002.37  4982.0 1998.42  4983.9 1996.42
  5010.8 1998.42  5014.8 2006.72  5022.9 2012.34  5087.2 2019.46  5257.3 2016.88
  5300.7 2012.96  5371.3 2013.58  5443.7 2004.90  5450.1 2006.51  5464.5 1999.72
  5499.8 2000.44  5520.6 2005.18  5564.1 2005.74  5671.8 2017.81  5803.2 2018.63
#Mann=7,-1,0
  2961.6    0.05       0  3817.1    0.12       0  4004.1    0.05       0
  4105.7    0.12       0  4318.7    0.05       0  4982.0    0.05       0
  5010.8    0.05       0
#XS Ineff=2,0
       0                 5097.70    0.00 2028.98
Permanent Ineff=
       F       F
Bank Sta=4982,5010.8
Exp/Cntr=0.3,0.1

Type RM Length L Ch R = 1,1012678,1075,1075,1075
BEGIN DESCRIPTION:
Clear Fork Brazos Rv 277.0
END DESCRIPTION:
XS GIS Cut Line= 4
      1329055.03      6970787.99      1330855.00      6970388.00
      1331239.59      6969955.33      1331326.45      6969551.43
#Sta/Elev= 30
  3155.1 2045.83  3247.3 2043.82  3462.4 2028.29  3579.2 2024.33  3725.0 2022.48
  3995.1 2017.89  4138.5 2018.15  4179.5 2016.17  4442.4 2016.10  4458.5 2016.50
  4882.4 2018.59  4958.0 2007.10  4968.2 2004.01  4979.8 1995.57  4983.1 1997.07
  4984.6 1995.07  5003.3 1995.07  5004.7 1997.07  5006.1 2006.01  5020.3 2008.19
  5091.4 2008.28  5154.9 2003.35  5175.8 1998.09  5183.4 1998.70  5190.1 2002.82
  5204.3 2005.29  5216.6 2010.27  5253.6 2015.61  5324.7 2018.30  5991.0 2018.21
#Mann=8,-1,0
  3155.1    0.05       0  3579.2    0.12       0  3725.0    0.05       0
  4442.4     0.1       0  4458.5    0.05       0  4983.1    0.05       0
  5004.7    0.05       0  5216.6    0.05       0
Bank Sta=4983.1,5004.7
Exp/Cntr=0.3,0.1

Type RM Length L Ch R = 1,1011603,298,298,298
BEGIN DESCRIPTION:
Mapping XS 9884f4c2
END DESCRIPTION:
XS GIS Cut Line= 6
      1330832.87      6974267.85      1331104.81      6973102.41
      1331289.03      6972312.92      1331677.19      6970780.01
      1331756.14      6970464.22      1332005.97      6969182.18
#Sta/Elev= 30
   986.3 2030.58  1848.7 2018.75  2772.9 2012.98  3102.0 2015.64  3153.6 2013.85
  3215.5 2002.78  3277.3 1999.13  3323.7 2004.18  3349.6 1999.15  3359.5 2004.34
  3370.2 1999.50  3390.8 2008.46  3419.6 2008.64  3569.7 2009.96  3586.8 1998.31
  3620.1 2009.72  3741.5 2014.36  4845.1 2016.40  4916.4 2009.56  4921.5 2012.92
  4968.0 2004.92  4973.1 2009.18  4988.4 2004.72  4997.5 1995.18  5001.4 1993.18
  5042.5 1995.18  5049.5 1993.68  5076.3 2004.33  5365.3 2016.87  6206.7 2017.32
#Mann=5,-1,0
   986.3    0.05       0  3419.6    0.12       0  3620.1    0.05       0
  4997.5    0.03       0  5042.5    0.05       0
#XS Ineff=2,0
    0.00 3704.50 2016.50               0
Permanent Ineff=
       F       F
Bank Sta=4997.5,5042.5
Exp/Cntr=0.3,0.1

Type RM Length L Ch R = 1,1011305,968,968,968
BEGIN DESCRIPTION:
Mapping XS 884ecbdb
END DESCRIPTION:
XS GIS Cut Line= 4
      1331169.05      6974347.87      1331387.98      6973248.85
      1331930.51      6970525.32      1332375.38      6968626.49
#Sta/Elev= 30
   760.3 2032.93  1843.1 2019.21  2910.8 2012.74  2966.9 2007.76  2983.0 2013.17
  3044.2 2000.54  3054.4 2001.36  3064.0 2007.21  3069.1 2004.86  3125.7 2013.62
  4790.5 2015.11  4870.3 2005.19  4953.1 2002.74  4960.4 1998.56  4965.5 1999.26
  4969.6 1994.77  4972.6 1992.77  5005.6 1994.77  5008.0 2006.91  5055.8 2015.80
  5220.1 2013.16  5400.4 2016.65  6041.8 2017.01  6185.2 2019.29  6232.8 2022.81
  6267.7 2020.74  6339.6 2025.85  6407.8 2025.27  6455.4 2029.24  6608.2 2031.61
#Mann=3,-1,0
   760.3    0.05       0  4969.6    0.03       0  5005.6    0.05       0
#XS Ineff=2,0
    0.00 3149.90 2015.76               0
Permanent Ineff=
       F       F
Bank Sta=4969.6,5005.6
Exp/Cntr=0.3,0.1

Type RM Length L Ch R = 1,1010337,1636,1636,1636
BEGIN DESCRIPTION:
Mapping XS f57cb7ff
END DESCRIPTION:
XS GIS Cut Line= 2
      1332494.75      6972934.18      1333058.99      6969027.92
#Sta/Elev= 30
  2627.2 2019.02  2855.7 2018.36  2886.0 2016.20  3078.0 2014.83  3229.6 2010.20
  3310.4 2011.17  3391.2 2003.21  3401.3 1997.13  3421.5 2003.18  3492.3 2011.95
  3967.1 2009.13  4856.3 2012.91  4917.4 2002.53  4972.4 2001.48  4977.0 1993.44
  4980.1 1991.44  5010.0 1991.44  5013.0 1993.44  5015.9 1998.88  5017.9 2002.63
  5028.0 2002.67  5058.4 2010.84  5078.6 2012.94  5605.4 2012.23  5715.1 2015.95
  6260.7 2019.22  6321.3 2022.47  6402.2 2021.85  6462.8 2025.67  6574.0 2025.93
#Mann=5,-1,0
  2627.2    0.05       0  4917.4     0.1       0  4977.0    0.07       0
  5013.0     0.1       0  5015.9    0.05       0
#XS Ineff=2,0
    0.00 3484.60 2014.23               0
Permanent Ineff=
       F       F
Bank Sta=4977,5013
Exp/Cntr=0.3,0.1

Type RM Length L Ch R = 1,1008701,2929,2929,2929
BEGIN DESCRIPTION:
Mapping XS 7ff4d2e6
END DESCRIPTION:
XS GIS Cut Line= 3
      1333178.34      6973129.51      1334148.72      6970123.36
      1333471.69      6968482.87
#Sta/Elev= 30
  1398.5 2020.63  1652.3 2018.72  1704.8 2014.78  1746.9 2015.99  1986.6 2007.77
  2413.6 2009.59  2461.4 2006.66  2482.9 1999.92  2509.7 1997.36  2515.0 1992.56
  2524.5 1997.37  2637.9 2009.59  3262.4 2006.65  4436.9 2009.73  4532.9 2013.87
  4885.4 2003.68  4958.9 1996.14  4971.2 1996.97  4983.9 1992.74  4986.2 1990.74
  5010.9 1992.74  5017.6 2004.66  5077.7 2006.40  5136.6 2012.39  5309.2 2012.28
  5391.8 2016.74  5666.6 2022.83  5759.2 2021.97  5836.4 2025.71  6332.1 2032.52
#Mann=5,-1,0
  1398.5    0.05       0  4885.4     0.1       0  4958.9    0.05       0
  4983.9    0.05       0  5010.9    0.05       0
#XS Ineff=2,0
    0.00 2640.40 2017.48 7359.60    0.00 2017.48
Permanent Ineff=
       F       F
Bank Sta=4983.9,5010.9
Exp/Cntr=0.3,0.1

Type RM Length L Ch R = 1,1005772,1320,1320,1320
BEGIN DESCRIPTION:
Clear Fork Brazos Rv 275.0
END DESCRIPTION:
XS GIS Cut Line= 3
      1333289.34      6972996.63      1334877.89      6971095.58
      1337605.03      6968537.97
#Sta/Elev= 30
  2535.5 2017.28  2908.0 2007.31  3368.7 2006.66  3419.4 1997.20  3425.9 1991.74
  3483.2 2007.48  3504.0 2008.05  4710.4 2006.82  4788.5 1996.84  4796.3 2001.60
  4817.1 2003.69  4866.6 1996.96  4938.1 1999.00  4981.1 1994.58  4981.4 1990.35
  4983.7 1988.35  5008.4 1990.35  5030.4 1988.45  5065.6 2001.70  5525.7 1999.89
  5596.5 2001.11  5645.8 2008.28  6005.3 2007.63  6233.0 2007.20  6260.5 2000.10
  7025.2 1999.27  7124.4 2002.69  7195.2 2010.83  8086.6 2014.00  8751.7 2030.79
#Mann=5,-1,0
  2535.5    0.05       0  4981.4    0.05       0  5008.4    0.05       0
  6005.3    0.12       0  6260.5    0.05       0
#XS Ineff=2,0
    0.00 3609.60 2008.44 5935.70    0.00 2015.50
Permanent Ineff=
       F       F
Bank Sta=4981.4,5008.4
Exp/Cntr=0.3,0.1

Type RM Length L Ch R = 1,1004452,2208,2208,2208
BEGIN DESCRIPTION:
Clear Fork Brazos Rv 274.0
END DESCRIPTION:
XS GIS Cut Line= 3
      1334278.95      6973369.86      1334851.85      6972232.73
      1338304.98      6968288.02
#Sta/Elev= 30
  3691.2 2021.98  4120.1 2009.27  4203.7 2002.58  4276.3 1992.24  4315.3 2000.50
  4382.2 2006.28  4850.7 2006.86  4902.6 1994.92  4947.4 1993.98  4956.7 1992.21
  4964.3 1986.10  4986.0 1987.72  4989.1 1985.72  5022.0 1987.72  5026.5 1995.73
  5040.7 1996.76  5154.6 1996.44  5310.3 2006.60  7017.7 2004.73  7301.5 2010.59
  7854.8 2008.00  8924.4 2015.26  9009.8 2013.17  9045.0 2016.63  9165.5 2017.11
  9278.4 2024.35  9300.3 2022.29  9555.6 2030.42  9916.2 2051.27 10207.1 2061.42
#Mann=3,-1,0
  3691.2    0.05       0  4986.0    0.05       0  5022.0    0.05       0
#XS Ineff=2,0
    0.00 4589.90 2009.13               0
Permanent Ineff=
       F       F
Bank Sta=4986,5022
Exp/Cntr=0.3,0.1

Type RM Length L Ch R = 1,1002244,1834,1834,1834
BEGIN DESCRIPTION:
Clear Fork Brazos Rv 273.0
END DESCRIPTION:
XS GIS Cut Line= 3
      1334804.97      6973288.02      1336596.64      6972232.73
      1338804.99      6969888.01
#Sta/Elev= 30
  2495.6 2023.81  2657.7 2020.96  2679.2 2012.92  2867.0 2014.46  2971.5 2006.47
  3006.3 1996.72  3056.2 1993.82  3073.5 1990.18  3079.3 1995.10  3190.7 1996.92
  3239.4 1990.56  3270.7 1998.45  3312.3 1995.18  3366.1 1988.82  3372.2 2000.94
  3393.6 2005.97  4561.4 2004.58  4754.0 1995.19  4914.9 1993.21  4982.9 1986.05
  4986.0 1984.05  5018.9 1986.05  5036.8 1994.03  5049.2 1993.69  5093.5 1993.01
  5143.2 2004.56  5645.3 2002.10  6925.9 2008.30  7449.4 2014.46  7795.9 2024.08
#Mann=7,-1,0
  2495.6    0.05       0  3056.2    0.12       0  3312.3    0.05       0
  4914.9     0.1       0  4982.9    0.07       0  5018.9     0.1       0
  5049.2    0.05       0
#XS Ineff=2,0
    0.00 4017.40 2006.47               0
Permanent Ineff=
       F       F
Bank Sta=4982.9,5018.9
Exp/Cntr=0.3,0.1

Type RM Length L Ch R = 1,1000410,934,934,934
BEGIN DESCRIPTION:
Clear Fork Brazos Rv 272.0
END DESCRIPTION:
XS GIS Cut Line= 3
      1335174.85      6973878.19      1336705.00      6973388.00
      1339404.98      6970388.03
#Sta/Elev= 30
  3385.6 2006.57  3426.0 2003.52  3466.3 2006.91  3774.3 2003.77  3879.3 1987.49
  3910.8 1997.16  3973.8 2003.46  4467.3 2002.38  4540.8 1998.44  4740.3 2001.63
  4855.8 1990.24  4971.0 1988.88  4981.8 1982.81  4984.8 1980.81  5017.8 1982.81
  5020.4 1988.03  5034.6 1990.44  5106.0 1991.43  5287.3 1986.39  5317.8 1992.68
  5343.5 1991.57  5374.7 1996.04  5530.5 1996.42  5608.6 2003.56  6868.8 2003.01
  7286.6 1998.31  7789.6 2006.83  8348.7 2008.04  8780.7 2016.50  9028.4 2028.97
#Mann=7,-1,0
  3385.6    0.12       0  3426.0    0.05       0  4981.8    0.07       0
  5017.8    0.05       0  5106.0    0.05       0  5287.3    0.12       0
  5343.5    0.05       0
#XS Ineff=2,0
    0.00 4660.10 2002.55               0
Permanent Ineff=
       F       F
Bank Sta=4981.8,5017.8
Exp/Cntr=0.3,0.1

Type RM Length L Ch R = 1,999476,1259,1259,1259
BEGIN DESCRIPTION:
Clear Fork Brazos Rv 271.0
END DESCRIPTION:
XS GIS Cut Line= 3
      1336845.87      6975505.80      1337555.00      6973338.00
      1339655.00      6970338.00
#Sta/Elev= 30
  2722.9 2016.17  3150.5 2010.42  3187.6 2007.61  3520.2 2001.48  4058.5 1998.73
  4162.0 2000.99  4625.0 2000.81  4732.9 1992.94  4987.8 1987.94  4991.7 1983.21
  4993.9 1981.21  5018.7 1983.21  5046.9 1989.48  5082.6 1993.13  5103.6 2001.92
  5383.4 1999.59  5499.4 2001.37  5556.1 1998.93  5785.4 2000.81  5844.7 1998.62
  6297.2 2001.35  6734.9 1997.70  6798.1 2001.51  6907.5 2001.05  7178.7 2006.71
  7345.2 2005.31  8012.2 2010.79  8306.9 2019.91  8348.8 2019.05  8665.7 2034.13
#Mann=3,-1,0
  2722.9    0.05       0  4991.7    0.07       0  5018.7    0.05       0
Bank Sta=4991.7,5018.7
Exp/Cntr=0.3,0.1

Type RM Length L Ch R = 1,998217,1589,1589,1589
BEGIN DESCRIPTION:
Clear Fork Brazos Rv 270.0
END DESCRIPTION:
XS GIS Cut Line= 3
      1337193.07      6975484.12      1338180.80      6974284.52
      1340405.02      6970037.96
#Sta/Elev= 30
  3389.8 2011.37  4482.8 1995.58  4830.7 2001.05  4974.9 1983.57  4977.9 1981.57
  5010.9 1983.57  5086.5 1987.76  5114.6 1993.34  5120.4 1998.76  5131.0 2002.45
  5390.1 1998.38  5506.1 2000.57  5572.3 1997.81  5707.4 2000.07  5775.1 1997.47
  5908.4 1999.45  6151.1 1996.68  7033.2 1996.80  7071.7 1999.25  7220.1 1998.28
  7441.2 2005.62  8337.7 2010.34  8507.0 2017.28  8543.9 2015.73  8654.2 2020.49
  9139.1 2028.54  9403.9 2038.06  9523.0 2046.01  9669.7 2047.59  9737.5 2052.41
#Mann=3,-1,0
  3389.8    0.05       0  4974.9    0.05       0  5010.9    0.05       0
Bank Sta=4974.9,5010.9
Exp/Cntr=0.3,0.1

Type RM Length L Ch R = 1,996628,1362,1362,1362
BEGIN DESCRIPTION:
Clear Fork Brazos Rv 269.0
END DESCRIPTION:
XS GIS Cut Line= 3
      1340187.02      6977065.07      1339447.88      6972771.06
      1340004.99      6971088.03
#Sta/Elev= 30
  1533.9 2015.82  1723.7 2014.60  1750.6 2011.10  2241.2 2003.50  2279.7 2000.80
  3529.9 1992.54  4676.5 1996.84  4700.7 1997.92  4717.1 2002.56  4778.0 1996.47
  4828.7 1985.99  4935.3 1985.16  4968.3 1980.34  4971.3 1978.34  5004.3 1980.34
  5011.4 1985.38  5062.1 1985.23  5194.0 1996.95  5298.0 1996.74  5764.0 1996.30
  5833.3 1993.47  5947.0 1997.44  6057.2 1996.38  6120.7 2000.23  6421.0 2006.23
  6968.7 2007.03  7221.5 2012.24  7262.3 2009.79  7547.7 2020.19  7663.9 2021.04
#Mann=4,-1,0
  1533.9    0.05       0  4968.3    0.07       0  5004.3    0.05       0
  5298.0    0.05       0
Bank Sta=4968.3,5004.3
Exp/Cntr=0.3,0.1

Type RM Length L Ch R = 1,995266,1219,1219,1219
BEGIN DESCRIPTION:
Clear Fork Brazos Rv 268.0
END DESCRIPTION:
XS GIS Cut Line= 2
      1340600.22      6976764.49      1340785.30      6972051.22
#Sta/Elev= 30
  1269.9 2008.25  1736.8 2001.49  1772.9 1999.06  2727.5 1996.83  3247.9 1991.45
  4348.8 1993.87  4388.8 1995.27  4418.8 2001.42  4458.8 1990.17  4488.9 1987.31
  4804.5 1983.07  4894.1 1982.18  4959.2 1984.32  4973.7 1980.25  4976.7 1978.25
  5006.7 1978.25  5009.7 1980.25  5049.3 1987.39  5069.3 1997.87  5094.1 1998.24
  5189.4 2005.78  5269.5 2003.93  5349.5 2008.47  5399.6 2007.52  5449.6 2012.07
  5489.6 2010.98  5699.8 2017.96  5739.8 2016.45  5809.9 2020.08  5986.8 2020.21
#Mann=6,-1,0
  1269.9    0.05       0  4804.5    0.12       0  4894.1    0.05       0
  4973.7    0.07       0  5009.7    0.05       0  5094.1    0.05       0
Bank Sta=4973.7,5009.7
Exp/Cntr=0.3,0.1

Type RM Length L Ch R = 1,994047,306,306,306
BEGIN DESCRIPTION:
Mapping XS e155350b
END DESCRIPTION:
XS GIS Cut Line= 3
      1341067.83      6976397.48      1341815.14      6973408.27
      1342164.82      6971971.73
#Sta/Elev= 30
  1638.4 2001.85  1815.3 2001.12  1851.3 1998.74  2122.3 1995.30  3500.6 1990.14
  4701.4 1993.17  4764.5 1997.08  4812.5 1994.00  4853.7 1984.26  4884.6 1981.65
  4989.2 1979.39  4992.2 1977.39  5022.2 1977.39  5025.2 1979.39  5028.6 1978.20
  5035.0 1980.78  5049.2 1981.81  5074.0 1989.18  5081.8 1992.92  5118.4 1995.42
  5234.5 1995.61  5255.1 1998.40  5290.5 1994.54  5843.2 1997.14  5926.6 1997.96
  5954.9 2000.18  6027.0 1998.81  6078.4 2002.24  6135.2 1999.98  6198.1 2004.16
#Mann=5,-1,0
  1638.4    0.05       0  4764.5    0.12       0  4989.2    0.07       0
  5025.2    0.12       0  5074.0    0.05       0
Bank Sta=4989.2,5025.2
Exp/Cntr=0.3,0.1

Type RM Length L Ch R = 1,993741,780,780,780
BEGIN DESCRIPTION:
Mapping XS a04bfabd
END DESCRIPTION:
XS GIS Cut Line= 3
      1341417.84      6976690.68      1342212.43      6972992.05
      1342429.64      6971821.04
#Sta/Elev= 30
  1457.4 2006.67  2339.8 1994.00  3083.9 1990.35  3182.6 1988.01  3301.2 1988.08
  3362.6 1990.60  4446.8 1991.04  4671.8 1992.27  4706.4 1993.07  4722.9 1996.02
  4763.8 1993.82  4794.5 1988.15  4844.3 1983.09  4927.5 1979.86  4987.3 1980.80
  4992.4 1977.48  4994.6 1975.48  5017.1 1975.48  5019.4 1977.48  5019.5 1975.98
  5080.9 1985.64  5121.8 1994.36  5661.1 1993.19  6058.2 1998.50  6139.6 2000.35
  6157.0 2003.53  6170.1 1999.89  6292.1 2006.59  6343.0 2004.79  6431.4 2007.62
#Mann=3,-1,0
  1457.4    0.05       0  4992.4    0.05       0  5019.4    0.05       0
Bank Sta=4992.4,5019.4
Exp/Cntr=0.3,0.1

Type RM Length L Ch R = 1,992961,933,933,933
BEGIN DESCRIPTION:
Clear Fork Brazos Rv 266.0
END DESCRIPTION:
XS GIS Cut Line= 3
      1342055.01      6977137.97      1342855.00      6973538.00
      1342647.56      6971478.51
#Sta/Elev= 30
  1317.5 2019.61  1754.1 2010.75  2003.8 2000.03  2280.4 1993.65  2957.8 1989.43
  3137.1 1986.01  3253.6 1985.79  3376.5 1989.70  4427.8 1989.46  4759.4 1993.31
  4790.2 1991.34  4810.7 1981.85  4840.1 1976.80  4937.4 1981.55  4956.2 1975.20
  4959.9 1973.20  5001.2 1975.20  5005.3 1980.82  5158.0 1982.84  5286.7 1992.94
  5497.8 1986.55  5889.7 1994.65  6362.1 1997.49  6382.2 2000.45  6422.4 1998.59
  6432.5 2000.55  6750.3 2001.58  6824.4 2006.15  6894.8 2004.94  7075.2 2008.76
#Mann=3,-1,0
  1317.5    0.05       0  4956.2    0.03       0  5001.2    0.05       0
#XS Ineff=2,0
    0.00 3690.10 1996.31               0
Permanent Ineff=
       F       F
Bank Sta=4956.2,5001.2
Exp/Cntr=0.3,0.1

Type RM Length L Ch R = 1,992028,1796,1796,1796
BEGIN DESCRIPTION:
Clear Fork Brazos Rv 265.0
END DESCRIPTION:
XS GIS Cut Line= 3
      1342155.01      6976887.98      1343655.00      6973888.00
      1343055.00      6970887.99
#Sta/Elev= 30
  1638.4 2014.24  1951.4 2003.71  2010.1 2004.90  2049.3 2000.99  2197.4 1996.83
  3248.3 1984.56  3539.0 1989.99  4760.5 1991.72  4782.8 1991.10  4844.3 1972.99
  4872.3 1978.39  4956.1 1980.32  4992.5 1977.98  4993.4 1973.28  4995.7 1971.28
  5020.4 1973.28  5023.1 1971.78  5043.5 1979.66  5114.9 1978.39  5216.8 1982.59
  5267.8 1991.37  5278.0 1988.58  5318.8 1992.76  6216.2 1991.80  6593.6 2000.77
  6614.0 1997.84  6654.8 2000.37  7664.4 2001.81  7776.5 2006.79  8051.9 2010.27
#Mann=3,-1,0
  1638.4    0.05       0  4993.4    0.05       0  5020.4    0.05       0
#XS Ineff=2,0
    0.00 4159.60 1993.40               0
Permanent Ineff=
       F       F
Bank Sta=4993.4,5020.4
Exp/Cntr=0.3,0.1

Type RM Length L Ch R = 1,990232,1920,1920,1920
BEGIN DESCRIPTION:
Mapping XS fafb45da
END DESCRIPTION:
XS GIS Cut Line= 3
      1343669.20      6976208.25      1344539.46      6974997.46
      1345692.84      6972331.45
#Sta/Elev= 30
  3919.1 1994.38  4130.5 1991.08  4746.8 1990.86  4811.8 1988.14  4868.3 1976.89
  4927.3 1976.44  4977.6 1975.85  4983.7 1974.34  4986.0 1970.52  4988.3 1968.52
  5013.0 1970.52  5013.2 1972.91  5034.0 1976.94  5057.8 1976.31  5335.6 1979.28
  5398.7 1977.52  5413.3 1979.84  5453.2 1976.20  5559.7 1979.50  5845.4 1974.63
  6062.1 1976.80  6281.3 1973.33  6318.8 1976.87  6342.3 1986.99  6488.3 1988.36
  6541.1 1984.97  7890.6 1986.59  7999.9 1987.21  8106.3 1995.54  8315.0 1992.55
#Mann=7,-1,0
  3919.1    0.05       0  4927.3    0.12       0  4986.0    0.07       0
  5013.0    0.12       0  5057.8    0.05       0  7890.6    0.12       0
  7999.9    0.05       0
Bank Sta=4986,5013
Exp/Cntr=0.3,0.1

Type RM Length L Ch R = 1,988312,922,922,922
BEGIN DESCRIPTION:
Clear Fork Brazos Rv 263.0
END DESCRIPTION:
XS GIS Cut Line= 3
      1345555.00      6976288.02      1345655.00      6975388.00
      1347454.99      6972388.02
#Sta/Elev= 30
  4093.3 1995.44  4193.9 1993.69  4244.2 1995.81  4264.4 1993.86  4566.2 1986.69
  4656.8 1978.45  4707.1 1983.69  4777.5 1973.85  4928.4 1972.63  4977.5 1965.42
  4980.5 1963.42  5010.5 1963.42  5013.5 1965.42  5022.2 1972.87  5043.6 1973.55
  5049.4 1977.72  5064.9 1982.17  5070.8 1986.67  5092.2 1989.26  5107.7 1986.88
  5166.0 1985.21  5626.7 1982.73  7529.5 1983.28  7615.0 1984.88  7622.8 1987.16
  7636.4 1984.86  7681.1 1987.30  8038.7 1988.16  8272.0 1993.30  8497.4 1995.39
#Mann=3,-1,0
  4093.3    0.05       0  4977.5    0.05       0  5013.5    0.05       0
Bank Sta=4977.5,5013.5
Exp/Cntr=0.3,0.1

Type RM Length L Ch R = 1,987390,931,931,931
BEGIN DESCRIPTION:
Clear Fork Brazos Rv 262.0
END DESCRIPTION:
XS GIS Cut Line= 4
      1345605.00      6976388.00      1346205.00      6976088.00
      1346642.43      6975650.57      1347717.74      6972038.37
#Sta/Elev= 30
  4329.4 1997.80  4471.9 1992.00  4634.1 1991.44  4919.2 1984.25  4941.5 1978.53
  4947.1 1973.77  4977.9 1971.48  4985.7 1966.15  4988.0 1964.15  5012.7 1966.15
  5014.4 1968.80  5028.5 1972.39  5110.2 1972.29  5162.6 1973.59  5184.1 1976.92
  5212.4 1986.51  5226.5 1987.08  5311.3 1982.24  5495.2 1981.89  8042.1 1983.46
  8156.9 1987.21  8188.2 1985.38  8203.9 1988.72  8237.1 1986.80  8479.7 1988.17
  9113.4 1998.09  9118.6 1995.94  9185.0 1998.50  9262.9 1996.60  9387.7 1998.33
#Mann=5,-1,0
  4329.4    0.05       0  4985.7    0.05       0  5012.7    0.05       0
  5110.2     0.1       0  5162.6    0.05       0
Bank Sta=4985.7,5012.7
Exp/Cntr=0.3,0.1

Type RM Length L Ch R = 1,986459,539,539,539
BEGIN DESCRIPTION:
Mapping XS 5fd769a9
END DESCRIPTION:
XS GIS Cut Line= 3
      1346610.96      6978379.55      1347027.63      6975996.70
      1347900.01      6972116.57
#Sta/Elev= 30
  3178.3 1996.09  3281.4 1993.07  3639.5 1992.25  4469.1 1982.45  4679.7 1984.59
  4804.1 1975.02  4986.9 1971.47  4991.7 1963.94  4993.9 1961.94  5016.4 1961.94
  5018.7 1963.94  5037.6 1969.99  5091.0 1971.25  5150.5 1983.18  5393.0 1981.08
  6754.2 1979.77  7194.9 1980.35  7328.2 1983.35  7410.2 1980.34  7520.3 1983.81
  8045.6 1983.65  8414.6 1986.54  8424.9 1988.90  9025.8 1991.09  9142.3 1992.51
  9173.1 1995.34  9203.8 1993.75  9408.8 1994.95  9436.0 1997.54  9574.3 1997.42
#Mann=3,-1,0
  3178.3    0.05       0  4991.7    0.05       0  5018.7    0.05       0
Bank Sta=4991.7,5018.7
Exp/Cntr=0.3,0.1

Type RM Length L Ch R = 1,985920,2048,2048,2048
BEGIN DESCRIPTION:
Clear Fork Brazos Rv 261.0
END DESCRIPTION:
XS GIS Cut Line= 3
      1346997.60      6978261.77      1347331.97      6976889.09
      1348898.24      6973756.55
#Sta/Elev= 30
  3530.2 1990.36  4275.1 1983.53  4686.8 1981.40  4903.0 1982.42  4931.7 1973.71
  4936.8 1973.96  4941.0 1970.97  4977.8 1967.96  4983.2 1965.41  4985.5 1963.41
  5008.0 1963.41  5010.2 1965.41  5011.3 1967.83  5033.7 1970.25  5139.9 1970.25
  5190.2 1974.11  5274.0 1974.89  5335.5 1983.41  5492.1 1980.33  6660.4 1977.58
  7353.6 1978.97  7487.7 1980.22  7510.1 1982.83  7594.0 1977.79  7717.0 1981.58
  7884.6 1981.37  7912.6 1983.45  8074.7 1979.21  8276.0 1980.15  8445.3 1985.84
#Mann=3,-1,0
  3530.2    0.05       0  4983.2    0.05       0  5010.2    0.05       0
Bank Sta=4983.2,5010.2
Exp/Cntr=0.3,0.1

Type RM Length L Ch R = 1,983872,1364,1364,1364
BEGIN DESCRIPTION:
Clear Fork Brazos Rv 260.0
END DESCRIPTION:
XS GIS Cut Line= 3
      1347457.35      6978801.77      1349056.62      6977505.03
      1349205.00      6973788.02
#Sta/Elev= 30
  1575.2 1991.53  3283.0 1986.08  3347.0 1983.67  3991.4 1979.30  4531.9 1978.70
  4561.9 1983.68  4652.0 1977.91  4772.1 1976.70  4822.1 1964.77  4832.9 1966.04
  4962.2 1967.29  4969.8 1964.46  4974.8 1965.56  4982.2 1962.61  4984.2 1959.58
  4986.4 1957.58  5008.9 1957.58  5011.2 1959.58  5012.3 1964.51  5022.3 1968.31
  5062.3 1978.41  5082.3 1980.23  5142.4 1978.10  5682.8 1977.38  6353.3 1981.28
  6477.5 1978.74  6483.4 1976.74  6663.6 1981.39  7013.8 1983.84  7354.1 1993.24
#Mann=4,-1,0
  1575.2    0.05       0  4832.9     0.1       0  4984.2    0.07       0
  5011.2    0.05       0
Bank Sta=4984.2,5011.2
Exp/Cntr=0.3,0.1

Type RM Length L Ch R = 1,982508,1758,1758,1758
BEGIN DESCRIPTION:
Clear Fork Brazos Rv 259.0
END DESCRIPTION:
XS GIS Cut Line= 3
      1347754.27      6978870.24      1349936.54      6977082.67
      1350854.99      6974988.02
#Sta/Elev= 30
  1039.7 1991.70  1304.6 1993.86  1325.4 1990.68  1362.0 1992.44  1809.2 1988.42
  2534.1 1986.71  3024.3 1980.88  3792.3 1977.70  3893.6 1974.84  4114.8 1978.47
  4219.2 1976.36  4378.9 1978.62  4440.5 1974.87  4661.8 1974.57  4706.5 1970.53
  4883.5 1967.19  4979.5 1964.22  4982.5 1957.37  4985.5 1955.37  5015.5 1955.37
  5018.5 1957.37  5023.2 1965.10  5045.1 1971.78  5077.8 1978.52  5094.6 1978.80
  5121.4 1980.69  5161.9 1977.11  5609.9 1980.24  5754.7 1972.74  6147.8 2002.00
#Mann=5,-1,0
  1039.7    0.05       0  4883.5     0.1       0  4982.5    0.07       0
  5018.5     0.1       0  5094.6    0.05       0
Bank Sta=4982.5,5018.5
Exp/Cntr=0.3,0.1

Type RM Length L Ch R = 1,980750,1150,1150,1150
BEGIN DESCRIPTION:
Mapping XS 45cf34ab
END DESCRIPTION:
XS GIS Cut Line= 4
      1349217.47      6978219.80      1350834.63      6977156.46
      1351454.90      6976713.41      1352052.61      6974831.75
#Sta/Elev= 30
  3392.1 1984.93  4171.0 1978.59  4705.6 1977.37  4806.7 1974.62  4838.0 1967.05
  4863.9 1961.03  4873.0 1963.61  4879.0 1961.51  4885.2 1965.00  4894.1 1965.90
  4980.9 1965.50  4982.0 1956.05  4985.0 1955.05  5018.0 1956.05  5023.6 1962.06
  5029.6 1964.09  5052.7 1963.93  5059.8 1960.13  5065.7 1959.91  5140.6 1965.99
  5318.8 1967.00  5413.7 1970.79  5470.2 1978.03  5915.1 1975.94  6036.7 1971.95
  6065.3 1975.45  6641.1 1972.50  7135.0 1973.38  7679.8 1982.00  8064.1 1994.41
#Mann=5,-1,0
  3392.1    0.05       0  4838.0    0.12       0  4982.0    0.07       0
  5018.0    0.12       0  5140.6    0.05       0
Bank Sta=4982,5018
Exp/Cntr=0.3,0.1

Type RM Length L Ch R = 1,979600,471,471,471
BEGIN DESCRIPTION:
Clear Fork Brazos Rv 258.0
END DESCRIPTION:
XS GIS Cut Line= 3
      1350957.25      6980479.15      1351643.59      6977417.04
      1352259.54      6974706.83
#Sta/Elev= 30
  1953.6 1986.44  2344.2 1982.38  3470.7 1977.35  4578.3 1974.17  4843.1 1976.67
  4865.2 1975.72  4891.6 1966.79  4906.2 1964.65  4957.5 1960.74  4967.7 1953.64
  4969.1 1955.14  4972.1 1953.14  5002.1 1953.14  5005.1 1955.14  5008.7 1961.57
  5031.9 1959.81  5075.3 1962.56  5093.8 1966.03  5118.5 1975.45  5161.5 1977.97
  5172.7 1975.82  5459.9 1974.90  5511.2 1970.51  5661.0 1977.04  5675.2 1974.55
  6167.5 1972.16  6936.6 1973.08  7149.0 1976.60  7439.1 1988.62  7871.0 2001.31
#Mann=3,-1,0
  1953.6    0.05       0  4969.1    0.05       0  5005.1    0.05       0
Bank Sta=4969.1,5005.1
Exp/Cntr=0.3,0.1

Type RM Length L Ch R = 1,979129,874,874,874
BEGIN DESCRIPTION:
Clear Fork Brazos Rv 257.0
END DESCRIPTION:
XS GIS Cut Line= 3
      1351274.02      6980549.56      1352065.95      6977610.62
      1352681.76      6974672.32
#Sta/Elev= 30
  1932.6 1983.75  2969.9 1980.59  3083.8 1975.89  4699.4 1973.24  4896.2 1975.36
  4918.6 1973.56  4953.3 1962.60  4989.3 1957.71  4992.5 1955.26  4994.7 1953.26
  5019.5 1955.26  5040.0 1959.18  5111.9 1963.17  5163.0 1975.08  5183.4 1976.15
  5520.6 1973.66  5602.3 1970.04  5778.6 1973.37  6777.3 1969.18  7053.1 1971.27
  7206.4 1976.99  7235.3 1980.49  7290.3 1980.33  7335.1 1984.43  7385.1 1983.42
  7429.9 1987.53  7502.7 1986.71  7574.2 1990.57  7679.5 1989.38  7978.5 1996.98
#Mann=3,-1,0
  1932.6    0.05       0  4992.5    0.03       0  5019.5    0.05       0
Bank Sta=4992.5,5019.5
Exp/Cntr=0.3,0.1

Type RM Length L Ch R = 1,978255,2050,2050,2050
BEGIN DESCRIPTION:
Clear Fork Brazos Rv 256.0
END DESCRIPTION:
XS GIS Cut Line= 3
      1352470.71      6980619.96      1352840.28      6977821.80
      1353473.83      6974988.43
#Sta/Elev= 30
  2146.4 1984.08  3025.9 1978.64  3530.3 1981.76  3641.2 1979.13  3746.0 1971.44
  3772.4 1973.85  3829.6 1967.03  3853.1 1962.39  3863.1 1966.32  3898.0 1967.10
  3925.4 1971.22  4105.2 1973.58  4760.9 1972.93  4801.2 1975.34  4851.7 1966.87
  4989.8 1955.29  4992.1 1953.29  5014.6 1953.29  5016.8 1955.29  5034.2 1959.18
  5075.2 1962.21  5116.2 1973.85  5146.4 1975.61  5208.4 1972.47  5310.9 1971.85
  5649.1 1974.51  5915.5 1970.00  6109.1 1971.71  6936.6 1967.03  7872.2 1977.51
#Mann=5,-1,0
  2146.4    0.05       0  3829.6    0.12       0  3925.4    0.05       0
  4989.8    0.05       0  5016.8    0.05       0
Bank Sta=4989.8,5016.8
Exp/Cntr=0.3,0.1

Type RM Length L Ch R = 1,976205,1856,1856,1856
BEGIN DESCRIPTION:
Clear Fork Brazos Rv 255.0
END DESCRIPTION:
XS GIS Cut Line= 3
      1353454.99      6981038.03      1354355.00      6978938.00
      1353849.98      6974088.79
#Sta/Elev= 30
  2722.6 1986.29  3803.3 1976.64  3843.2 1980.24  4254.9 1972.73  4671.1 1971.24
  4788.0 1970.50  4811.5 1962.39  4822.4 1968.19  4833.3 1967.57  4864.1 1961.96
  4869.6 1964.91  4945.7 1956.36  4967.9 1951.02  4970.9 1949.02  5003.9 1951.02
  5004.6 1955.72  5101.4 1958.57  5238.6 1963.79  5298.9 1971.12  5459.8 1966.70
  8274.9 1967.30  8821.8 1972.99  8988.8 1969.29  9159.7 1978.47  9230.1 1978.36
  9250.2 1986.91  9260.2 1982.89  9304.4 1981.73  9481.4 1989.47  9882.8 1996.23
#Mann=5,-1,0
  2722.6    0.05       0  4671.1    0.12       0  4967.9    0.07       0
  5003.9    0.12       0  5101.4    0.05       0
Bank Sta=4967.9,5003.9
Exp/Cntr=0.3,0.1

Type RM Length L Ch R = 1,974349,1175,1175,1175
BEGIN DESCRIPTION:
Clear Fork Brazos Rv 254.0
END DESCRIPTION:
XS GIS Cut Line= 3
      1355219.19      6979906.88      1355255.00      6977738.00
      1354992.27      6974941.89
#Sta/Elev= 30
  2823.0 1972.69  3041.9 1971.29  3081.9 1969.22  4142.1 1967.48  4162.1 1963.73
  4232.1 1959.18  4832.2 1960.42  4913.1 1958.92  4952.2 1957.37  4982.2 1952.55
  4986.9 1947.71  4989.9 1945.71  5019.9 1945.71  5022.9 1947.71  5032.4 1952.48
  5078.4 1957.38  5122.7 1958.06  5132.8 1959.45  5150.2 1966.25  5162.9 1967.71
  5173.0 1965.34  5193.1 1965.12  6629.4 1964.45  7151.6 1966.73  7533.3 1971.82
  7573.5 1974.27  7614.9 1972.42  7663.9 1976.15  7718.6 1974.86  7800.6 1976.78
#Mann=5,-1,0
  2823.0    0.05       0  4913.1    0.12       0  4986.9    0.07       0
  5022.9    0.12       0  5078.4    0.05       0
Bank Sta=4986.9,5022.9
Exp/Cntr=0.3,0.1

Type RM Length L Ch R = 1,973174,1439,1439,1439
BEGIN DESCRIPTION:
Clear Fork Brazos Rv 252.0
END DESCRIPTION:
XS GIS Cut Line= 3
      1356240.81      6980550.14      1356205.00      6978288.00
      1355862.46      6975432.80
#Sta/Elev= 30
  2735.9 1979.20  2768.0 1982.17  2808.1 1979.53  3688.2 1967.62  4708.3 1966.56
  4798.3 1957.75  4938.3 1956.95  4959.8 1954.88  4988.3 1950.70  4989.4 1948.65
  4992.4 1946.65  5022.4 1946.65  5025.4 1948.65  5048.7 1952.04  5078.9 1952.17
  5099.0 1949.55  5140.8 1956.21  5210.3 1960.41  5250.1 1967.28  5416.3 1967.99
  5471.7 1968.09  5501.9 1964.40  6408.4 1962.07  6458.7 1964.14  6529.2 1961.62
  6861.6 1961.71  7083.2 1964.26  7606.9 1964.87  7798.3 1969.83  7874.0 1968.99
#Mann=7,-1,0
  2735.9    0.05       0  4959.8    0.12       0  4989.4    0.07       0
  5025.4    0.12       0  5140.8    0.05       0  5210.3    0.12       0
  5416.3    0.05       0
Bank Sta=4989.4,5025.4
Exp/Cntr=0.3,0.1

Type RM Length L Ch R = 1,971735,1673,1673,1673
BEGIN DESCRIPTION:
Clear Fork Brazos Rv 251.0
END DESCRIPTION:
XS GIS Cut Line= 3
      1356534.05      6980238.00      1357155.14      6977346.33
      1357347.44      6975471.68
#Sta/Elev= 30
  2040.9 1975.51  2546.3 1968.54  4188.8 1964.28  4250.2 1966.54  4291.1 1961.64
  4761.6 1957.92  4822.9 1953.81  4863.8 1955.53  4893.2 1951.50  4960.6 1947.62
  4964.3 1945.62  5005.6 1947.62  5006.9 1951.19  5016.9 1951.87  5097.4 1951.28
  5137.1 1955.56  5177.8 1963.39  5268.3 1960.64  5298.4 1964.64  5308.5 1960.97
  5368.8 1960.41  6324.4 1960.08  6494.7 1961.88  6517.9 1969.58  6544.9 1965.13
  6575.1 1967.61  6735.9 1965.90  6836.4 1969.43  6846.5 1974.56  6883.0 1971.64
#Mann=5,-1,0
  2040.9    0.05       0  4893.2    0.12       0  4960.6    0.07       0
  5005.6    0.12       0  5137.1    0.05       0
Bank Sta=4960.6,5005.6
Exp/Cntr=0.3,0.1

Type RM Length L Ch R = 1,970062,1279,1279,1279
BEGIN DESCRIPTION:
Clear Fork Brazos Rv 250.0
END DESCRIPTION:
XS GIS Cut Line= 3
      1357565.14      6980550.16      1357970.61      6978502.44
      1358255.50      6975321.05
#Sta/Elev= 30
  2932.3 1982.91  3219.9 1979.83  3260.7 1976.91  3505.4 1972.68  3974.3 1970.36
  4449.5 1963.67  4472.9 1963.69  4535.0 1961.80  4639.1 1953.15  4864.2 1953.17
  4891.8 1950.54  4973.3 1952.93  4983.5 1952.26  4996.8 1945.90  4997.5 1944.90
  5005.8 1945.90  5024.5 1948.95  5094.2 1950.39  5395.7 1953.12  5461.2 1961.82
  5625.3 1961.39  6160.8 1959.89  6263.9 1959.31  7316.9 1960.11  7320.7 1960.17
  7504.2 1961.25  7813.1 1973.82  7875.6 1972.57  8152.0 1981.35  8213.9 1980.81
#Mann=13,-1,0
  2932.3    0.05       0  4449.5    0.12       0  4472.9    0.05       0
  4639.1    0.12       0  4996.8    0.07       0  5005.8    0.12       0
  5094.2    0.05       0  5625.3    0.12       0  6160.8    0.05       0
  6263.9    0.12       0  7316.9    0.05       0  7320.7    0.12       0
  7504.2    0.05       0
Bank Sta=4996.8,5005.8
Exp/Cntr=0.3,0.1

Type RM Length L Ch R = 1,968783,1847,1847,1847
BEGIN DESCRIPTION:
Clear Fork Brazos Rv 249.0
END DESCRIPTION:
XS GIS Cut Line= 3
      1358855.00      6980638.03      1358855.00      6977938.00
      1358555.00      6974937.99
#Sta/Elev= 30
  2310.1 1984.79  3040.1 1969.26  3923.6 1962.56  4080.6 1961.75  4305.5 1962.46
  4390.1 1951.02  4510.8 1950.00  4650.1 1951.83  4760.1 1947.25  4800.1 1950.54
  4896.0 1951.00  4970.1 1947.29  4988.8 1943.81  4991.0 1942.81  5015.8 1943.81
  5057.9 1952.07  5062.9 1949.88  5070.4 1953.40  5098.7 1956.10  5344.9 1957.41
  6588.0 1955.81  6799.0 1956.71  6988.0 1963.75  7168.3 1975.70  7201.0 1972.58
  7369.3 1979.61  7532.6 1980.58  7904.5 1988.75  7954.7 1992.01  8025.1 1991.05
#Mann=11,-1,0
  2310.1    0.05       0  3923.6    0.12       0  4080.6    0.05       0
  4305.5    0.12       0  4510.8    0.05       0  4896.0    0.12       0
  4988.8    0.07       0  5015.8    0.12       0  5098.7    0.05       0
  5344.9    0.12       0  6988.0    0.05       0
Bank Sta=4988.8,5015.8
Exp/Cntr=0.3,0.1

Type RM Length L Ch R = 1,966936,918,918,918
BEGIN DESCRIPTION:
Clear Fork Brazos Rv 248.0
END DESCRIPTION:
XS GIS Cut Line= 3
      1359604.99      6980188.02      1360405.00      6978788.00
      1358805.01      6975188.01
#Sta/Elev= 30
  3367.6 1977.21  3918.3 1965.79  4500.9 1959.81  4680.6 1959.96  4876.4 1944.90
  4885.8 1947.87  4982.8 1946.47  4994.4 1946.23  4996.9 1942.61  4999.2 1941.61
  5023.9 1942.61  5104.1 1946.22  5168.2 1950.74  5321.0 1949.99  5410.3 1950.44
  5510.1 1952.32  5588.0 1960.16  6557.1 1956.00  6734.9 1955.87  7055.9 1955.07
  7106.9 1955.36  7153.3 1955.10  7638.1 1954.52  7711.9 1954.53  8016.2 1962.30
  8031.9 1963.12  8131.7 1969.39  8175.5 1968.10  8350.6 1975.41  8919.6 1987.08
#Mann=17,-1,0
  3367.6    0.05       0  4500.9    0.12       0  4996.9    0.03       0
  5023.9    0.05       0  5104.1    0.05       0  5321.0    0.12       0
  5410.3    0.05       0  5588.0    0.12       0  6557.1    0.05       0
  6734.9    0.12       0  7055.9    0.05       0  7106.9    0.12       0
  7153.3    0.05       0  7638.1    0.12       0  7711.9    0.05       0
  8016.2    0.12       0  8031.9    0.05       0
Bank Sta=4996.9,5023.9
Exp/Cntr=0.3,0.1

Type RM Length L Ch R = 1,966018,2786,2786,2786
BEGIN DESCRIPTION:
Clear Fork Brazos Rv 247.0
END DESCRIPTION:
XS GIS Cut Line= 3
      1361205.00      6980938.05      1361205.00      6978938.00
      1358805.01      6974938.01
#Sta/Elev= 30
  2994.5 1985.37  3414.5 1974.34  3474.5 1974.99  3594.5 1969.94  3974.5 1963.70
  4844.5 1960.48  4901.2 1956.04  4924.5 1948.33  4984.5 1945.44  4989.0 1941.37
  4991.2 1940.37  5016.0 1941.37  5017.9 1943.52  5066.5 1947.62  5303.2 1945.81
  5358.0 1945.95  5437.7 1958.50  5461.0 1958.89  6219.0 1955.06  7019.9 1955.07
  7273.7 1954.99  7368.0 1954.68  8018.9 1953.26  8326.0 1961.41  8458.1 1970.44
  8506.7 1966.93  8691.4 1975.45  9367.8 1984.40  9556.3 1991.47  9659.3 1992.34
#Mann=8,-1,0
  2994.5    0.05       0  4901.2    0.12       0  4989.0    0.07       0
  5016.0    0.12       0  5303.2    0.12       0  7019.9    0.05       0
  7273.7    0.12       0  7368.0    0.05       0
Bank Sta=4989,5016
Exp/Cntr=0.3,0.1
