HEC-RAS study Clear Fork Brazos Rv.prj: Clear Fork Brazos Rv Base Level Engineering

--- Clear Fork Brazos Rv.g01 (geometry) --- (continued)

Type RM Length L Ch R = 1,828770,3220,3220,3220
BEGIN DESCRIPTION:
Clear Fork Brazos Rv 193.0
END DESCRIPTION:
XS GIS Cut Line= 3
      1432655.00      6958788.01      1430155.00      6953788.00
      1428654.98      6951287.96
#Sta/Elev= 30
  -589.4 1880.08  -402.1 1880.94     0.4 1867.73   268.7 1868.30   671.2 1846.95
  1029.0 1838.44  3919.1 1840.00  4226.5 1835.13  4643.0 1837.64  4701.7 1833.60
  4917.0 1836.88  4970.0 1833.64  4984.2 1825.18  4986.5 1824.18  5011.2 1825.18
  5045.5 1836.13  5150.8 1833.67  5247.6 1838.24  6143.6 1838.46  6190.3 1832.77
  6248.6 1837.81  6575.1 1840.32  6715.1 1850.52  6843.4 1850.28  6917.2 1842.31
  6948.3 1849.21  7028.0 1851.47  7055.2 1848.58  7325.4 1856.69  7916.3 1860.84
#Mann=5,-1,0
  -589.4    0.05       0  4917.0    0.12       0  4984.2    0.07       0
  5011.2    0.12       0  5150.8    0.05       0
Bank Sta=4984.2,5011.2
Exp/Cntr=0.3,0.1

Type RM Length L Ch R = 1,825550,614,614,614
BEGIN DESCRIPTION:
Mapping XS 6db7db48
END DESCRIPTION:
XS GIS Cut Line= 4
      1435320.45      6958301.42      1432750.99      6954811.82
      1431275.30      6951999.32      1429365.56      6950454.17
#Sta/Elev= 30
 -1884.6 1851.46 -1849.7 1856.07 -1805.8 1858.07 -1784.9 1857.15 -1728.6 1848.70
  -849.2 1843.14  -203.9 1843.16  1590.5 1836.97  2398.9 1836.89  2818.6 1839.67
  3358.7 1835.31  4306.5 1834.95  4344.9 1831.65  4395.6 1835.43  4521.4 1834.00
  4863.0 1835.90  4892.5 1832.21  4945.5 1832.12  4960.3 1829.51  4967.6 1823.98
  4981.3 1822.93  4983.6 1821.93  5008.3 1822.93  5011.7 1831.43  5077.8 1836.84
  5726.2 1834.16  6429.7 1834.98  6578.4 1840.46  6990.9 1849.90  8081.6 1856.65
#Mann=3,-1,0
 -1884.6    0.05       0  4981.3    0.05       0  5008.3    0.05       0
Bank Sta=4981.3,5008.3
Exp/Cntr=0.3,0.1

Type RM Length L Ch R = 1,824936,1807,1807,1807
BEGIN DESCRIPTION:
Mapping XS e73d3253
END DESCRIPTION:
XS GIS Cut Line= 4
      1434973.23      6956218.08      1433150.30      6954169.46
      1432004.46      6952311.82      1430216.55      6950072.59
#Sta/Elev= 30
   392.4 1854.78   639.0 1852.06   844.7 1862.60  1021.6 1852.00  1341.7 1843.82
  1396.5 1842.74  2197.7 1832.41  2261.2 1838.16  2296.3 1831.85  2339.0 1838.27
  2558.9 1837.65  2594.0 1833.74  2707.7 1838.13  2728.6 1834.43  2757.1 1839.22
  2834.8 1835.16  3047.2 1835.01  3134.7 1839.34  4615.9 1827.70  4832.3 1830.15
  4969.5 1829.27  4984.9 1826.44  4986.6 1822.01  4988.8 1821.01  5013.6 1822.01
  5037.0 1832.25  5051.5 1833.67  6550.6 1830.04  6977.2 1842.12  8182.7 1848.37
#Mann=5,-1,0
   392.4    0.05       0  1341.7    0.12       0  1396.5    0.05       0
  4986.6    0.03       0  5013.6    0.05       0
Bank Sta=4986.6,5013.6
Exp/Cntr=0.3,0.1

Type RM Length L Ch R = 1,823129,1577,1577,1577
BEGIN DESCRIPTION:
Mapping XS 6ec5b9ac
END DESCRIPTION:
XS GIS Cut Line= 3
      1435763.95      6954857.86      1432777.86      6951472.47
      1430399.66      6949979.58
#Sta/Elev= 30
   586.4 1846.09  1499.5 1834.76  2519.7 1829.46  2931.0 1830.71  3164.3 1828.82
  3596.9 1831.43  4297.9 1831.95  4397.5 1828.58  4574.0 1831.59  4886.1 1831.52
  4949.7 1833.11  4963.9 1830.61  4971.4 1826.37  4974.0 1821.10  4977.0 1820.10
  5010.0 1821.10  5013.2 1827.54  5020.8 1829.10  5141.2 1834.36  5925.8 1831.48
  6245.1 1828.25  6579.7 1835.37  6709.7 1840.02  6983.8 1840.32  6999.1 1842.17
  7202.9 1842.57  7260.6 1844.65  7339.6 1842.48  7360.8 1844.43  7908.5 1848.22
#Mann=3,-1,0
   586.4    0.05       0  4974.0    0.05       0  5010.0    0.05       0
Bank Sta=4974,5010
Exp/Cntr=0.3,0.1

Type RM Length L Ch R = 1,821552,5438,5438,5438
BEGIN DESCRIPTION:
Clear Fork Brazos Rv 190.0
END DESCRIPTION:
XS GIS Cut Line= 3
      1436505.02      6954238.02      1433505.00      6950238.00
      1430004.96      6949737.99
#Sta/Elev= 30
    -0.1 1873.20   192.6 1871.93   307.2 1859.74   342.6 1862.85   413.5 1860.42
   442.6 1850.71   478.1 1847.14  1128.1 1832.39  2013.5 1828.26  3263.5 1830.55
  3607.2 1825.48  3757.2 1828.55  4878.1 1832.56  4936.4 1829.91  4966.6 1821.20
  4970.3 1820.20  5011.6 1821.20  5020.1 1829.44  5030.2 1831.18  5121.1 1829.81
  5191.9 1833.77  5626.2 1831.01  6808.1 1832.01  6989.9 1837.67  7353.6 1839.95
  7424.3 1841.94  7434.4 1844.84  7484.9 1839.22  7606.1 1843.72  8535.5 1854.16
#Mann=3,-1,0
    -0.1    0.05       0  4966.6    0.05       0  5011.6    0.05       0
Bank Sta=4966.6,5011.6
Exp/Cntr=0.3,0.1

Type RM Length L Ch R = 1,816114,4065,4065,4065
BEGIN DESCRIPTION:
Clear Fork Brazos Rv 189.0
END DESCRIPTION:
XS GIS Cut Line= 3
      1436855.00      6953487.99      1433961.25      6948692.17
      1432354.98      6944987.96
#Sta/Elev= 30
  -609.6 1871.30  -586.3 1868.47  -543.6 1854.90  -368.9 1844.64  -142.4 1837.19
   345.4 1830.51  2092.4 1823.76  4342.4 1827.86  4685.7 1824.66  4961.5 1828.41
  4976.8 1824.70  4993.0 1812.98  4995.3 1811.98  5020.0 1812.98  5045.1 1817.30
  5061.6 1824.85  5092.1 1828.17  5547.2 1827.55  5576.1 1833.44  5617.5 1824.65
  5737.3 1824.46  6336.8 1832.31  6726.5 1832.95  6794.6 1839.66  6831.2 1836.02
  7105.7 1835.62  8162.2 1845.10  8891.8 1854.72  8915.3 1858.24  9029.1 1854.80
#Mann=3,-1,0
  -609.6    0.05       0  4993.0    0.05       0  5020.0    0.05       0
Bank Sta=4993,5020
Exp/Cntr=0.3,0.1

Type RM Length L Ch R = 1,812049,3108,3108,3108
BEGIN DESCRIPTION:
Clear Fork Brazos Rv 188.0
END DESCRIPTION:
XS GIS Cut Line= 3
      1437560.01      6952554.86      1435305.00      6947438.00
      1433168.82      6945194.98
#Sta/Elev= 30
  -591.6 1848.27  -398.5 1836.29  -288.8 1833.08   948.6 1829.28  1912.9 1822.33
  2185.9 1823.08  2255.9 1821.02  2284.7 1822.76  2923.8 1822.81  3155.7 1824.94
  3371.2 1822.92  4764.9 1825.32  4863.6 1823.10  4939.1 1824.24  4967.9 1820.61
  4978.3 1816.88  4983.9 1811.16  4986.1 1810.16  5010.9 1811.16  5014.1 1820.06
  5021.4 1824.11  5049.7 1826.62  5368.0 1821.79  5608.3 1821.99  5658.0 1825.03
  5884.1 1828.76  5948.0 1831.78  6167.2 1834.36  7171.5 1839.17  8097.6 1849.49
#Mann=3,-1,0
  -591.6    0.05       0  4983.9    0.05       0  5010.9    0.05       0
Bank Sta=4983.9,5010.9
Exp/Cntr=0.3,0.1

Type RM Length L Ch R = 1,808941,4084,4084,4084
BEGIN DESCRIPTION:
Mapping XS 9e3c1745
END DESCRIPTION:
XS GIS Cut Line= 3
      1439210.52      6951656.08      1437023.01      6947281.06
      1434385.00      6945042.23
#Sta/Elev= 30
   361.0 1861.60   424.8 1861.75   519.8 1855.47   670.8 1852.33   872.0 1841.65
   996.1 1837.45  1443.3 1827.37  1766.4 1824.89  2325.5 1825.28  2912.4 1819.38
  3041.0 1821.18  4919.3 1822.56  4969.6 1819.63  4987.7 1810.77  4990.7 1809.77
  5023.7 1810.77  5031.1 1816.15  5036.7 1816.22  5043.4 1820.85  5059.0 1822.68
  5480.3 1819.38  6040.5 1821.91  6076.1 1820.45  6089.9 1822.68  6167.9 1820.42
  6813.7 1820.73  6906.0 1818.10  7125.7 1824.48  7715.6 1831.79  8712.4 1836.47
#Mann=3,-1,0
   361.0    0.05       0  4987.7    0.05       0  5023.7    0.05       0
Bank Sta=4987.7,5023.7
Exp/Cntr=0.3,0.1

Type RM Length L Ch R = 1,804857,2599,2599,2599
BEGIN DESCRIPTION:
Clear Fork Brazos Rv 187.0
END DESCRIPTION:
XS GIS Cut Line= 3
      1442664.16      6948856.94      1440105.00      6947288.00
      1435424.58      6943735.41
#Sta/Elev= 30
  1997.6 1843.24  2315.2 1838.13  2794.8 1837.80  3632.2 1832.65  4090.5 1827.96
  4301.3 1823.00  4359.3 1824.57  4649.4 1818.70  4846.9 1817.20  4970.4 1818.84
  4985.8 1818.34  4993.0 1807.93  4996.0 1806.93  5029.0 1807.93  5035.8 1809.83
  5042.1 1817.36  5071.2 1820.15  5313.3 1816.39  6462.6 1817.21  6776.7 1813.64
  6847.4 1817.07  7246.8 1817.89  8218.0 1816.09  9074.9 1817.65  9131.1 1819.95
  9788.3 1818.21  9988.0 1822.16 10109.1 1829.22 10209.5 1830.60 10875.4 1830.44
#Mann=3,-1,0
  1997.6    0.05       0  4993.0    0.05       0  5029.0    0.05       0
Bank Sta=4993,5029
Exp/Cntr=0.3,0.1

Type RM Length L Ch R = 1,802258,2178,2178,2178
BEGIN DESCRIPTION:
Clear Fork Brazos Rv 186.0
END DESCRIPTION:
XS GIS Cut Line= 3
      1443044.57      6947233.82      1442044.58      6946213.00
      1435233.06      6940172.20
#Sta/Elev= 30
  3559.6 1830.55  4652.4 1823.09  4765.6 1820.77  4800.9 1816.49  4822.1 1819.55
  4829.1 1814.78  4836.3 1815.98  4850.4 1812.72  4899.9 1812.20  4907.0 1813.93
  4914.0 1811.53  4942.3 1812.23  4970.6 1809.58  4981.9 1806.62  4984.2 1805.62
  5008.9 1806.62  5013.4 1814.60  5055.2 1817.04  7591.8 1814.37  7641.2 1809.27
  7669.6 1814.77  8654.0 1812.00 11615.5 1821.77 12175.0 1827.24 12720.2 1838.81
 12911.8 1836.14 13130.9 1838.48 13350.8 1836.04 13655.3 1839.98 14092.9 1839.00
#Mann=3,-1,0
  3559.6    0.05       0  4981.9    0.05       0  5008.9    0.05       0
Bank Sta=4981.9,5008.9
Exp/Cntr=0.3,0.1

Type RM Length L Ch R = 1,800080,2397,2397,2397
BEGIN DESCRIPTION:
Clear Fork Brazos Rv 185.0
END DESCRIPTION:
XS GIS Cut Line= 3
      1444405.01      6945838.00      1442405.00      6944338.00
      1434404.96      6937337.97
#Sta/Elev= 30
  2505.4 1852.32  2905.4 1849.45  2918.9 1847.15  3220.9 1831.02  3305.4 1825.58
  4248.1 1813.30  4416.1 1814.40  4605.4 1815.64  4705.4 1813.10  4948.1 1815.09
  4968.9 1805.65  4979.7 1805.18  4981.9 1804.18  5006.7 1805.18  5008.7 1815.59
  5033.4 1816.38  6982.9 1811.27  7003.8 1809.69  7038.9 1811.60  7053.1 1810.00
  7075.0 1812.47  7103.4 1808.51  7124.3 1808.30  7159.4 1811.20  7251.5 1812.28
 11064.6 1825.94 13389.5 1842.26 14289.2 1853.28 14798.9 1863.55 15635.6 1864.75
#Mann=5,-1,0
  2505.4    0.05       0  3220.9    0.12       0  4416.1    0.05       0
  4979.7    0.05       0  5006.7    0.05       0
Bank Sta=4979.7,5006.7
Exp/Cntr=0.3,0.1

Type RM Length L Ch R = 1,797683,4767,4767,4767
BEGIN DESCRIPTION:
Clear Fork Brazos Rv 184.0
END DESCRIPTION:
XS GIS Cut Line= 3
      1444554.99      6944737.99      1444055.00      6944238.00
      1435054.96      6937237.97
#Sta/Elev= 30
  4280.5 1841.74  4735.2 1835.67  4775.2 1834.95  4888.6 1831.72  4931.0 1826.29
  4984.9 1804.88  4987.2 1803.78  5011.9 1804.88  5059.1 1812.70  7132.2 1815.27
  8073.3 1808.16  8102.3 1810.91  8172.8 1805.97  8201.8 1811.38 11258.6 1816.97
 12406.0 1828.61 12441.3 1833.77 12520.0 1826.20 12590.6 1830.81 14628.4 1847.13
 15121.6 1856.94 15241.9 1864.70 15384.9 1861.04 15505.3 1870.06 15741.4 1867.97
 15905.2 1875.54 16060.9 1869.46 16098.0 1876.62 16197.5 1876.44 16389.4 1866.42
#Mann=5,-1,0
  4280.5    0.05       0  4735.2    0.12       0  4775.2    0.05       0
  4984.9    0.05       0  5011.9    0.05       0
Bank Sta=4984.9,5011.9
Exp/Cntr=0.3,0.1

Type RM Length L Ch R = 1,792916,3406,3406,3406
BEGIN DESCRIPTION:
Clear Fork Brazos Rv 183.0
END DESCRIPTION:
XS GIS Cut Line= 3
      1445704.97      6944787.97      1441705.00      6940788.00
      1437205.03      6938288.02
#Sta/Elev= 30
  -651.1 1850.48    13.5 1839.32    98.4 1835.98   140.8 1829.91   282.2 1825.98
   324.7 1828.30   480.2 1825.87   522.7 1832.59   565.1 1828.94   961.1 1812.37
  2219.7 1809.46  3252.1 1811.43  3973.3 1808.19  4722.9 1810.85  4892.6 1806.04
  4935.0 1808.38  4963.3 1800.09  4973.0 1799.66  4976.0 1798.66  5009.0 1799.66
  5013.7 1809.89  5041.2 1814.12  5078.9 1811.44  5350.0 1810.30  5999.8 1811.71
  7896.5 1820.98  8953.5 1831.62  9787.5 1847.98 10036.8 1861.40 10153.5 1858.79
#Mann=3,-1,0
  -651.1    0.05       0  4973.0    0.05       0  5009.0    0.05       0
Bank Sta=4973,5009
Exp/Cntr=0.3,0.1

Type RM Length L Ch R = 1,789510,11210,11210,11210
BEGIN DESCRIPTION:
Mapping XS 0e8baea5
END DESCRIPTION:
XS GIS Cut Line= 4
      1445650.31      6944308.38      1444296.13      6941981.96
      1442125.99      6939325.71      1437978.32      6938180.33
#Sta/Elev= 30
  1769.1 1842.22  1884.2 1840.15  1911.5 1843.49  1933.0 1840.52  2007.5 1842.26
  2044.7 1839.49  2081.9 1830.31  2301.2 1831.43  2313.4 1828.48  2403.0 1822.92
  2569.3 1819.80  2695.2 1812.29  2782.7 1810.78  4460.3 1806.79  4912.4 1808.95
  4926.7 1806.90  4933.2 1798.90  4941.1 1799.39  4955.3 1795.23  4959.0 1794.23
  5000.3 1795.23  5005.0 1804.82  5011.4 1806.51  5118.4 1804.50  5217.5 1807.37
  6916.8 1805.25  7306.9 1808.54  8722.0 1811.48 10151.8 1819.54 12193.9 1837.00
#Mann=3,-1,0
  1769.1    0.05       0  4955.3    0.05       0  5000.3    0.05       0
Bank Sta=4955.3,5000.3
Exp/Cntr=0.3,0.1

Type RM Length L Ch R = 1,778300,4448,4448,4448
BEGIN DESCRIPTION:
Mapping XS 1c867b80
END DESCRIPTION:
XS GIS Cut Line= 3
      1448619.07      6941131.28      1446211.25      6939525.50
      1442560.01      6934985.41
#Sta/Elev= 30
  1801.3 1831.76  2340.0 1826.36  2982.9 1804.58  3869.2 1803.11  4100.6 1800.83
  4762.1 1802.20  4875.6 1797.85  4974.8 1796.05  4989.2 1797.26  4990.0 1788.85
  4992.2 1787.95  5017.0 1788.85  5025.9 1791.51  5032.4 1798.86  5075.6 1802.88
  5835.6 1801.81  6462.7 1803.41  6533.1 1795.80  6568.3 1801.11  6739.5 1801.10
  6888.3 1804.45  6931.5 1802.45  6995.5 1804.58  7045.1 1803.02  8155.3 1803.42
  8432.1 1806.51  8859.3 1806.93  9548.8 1813.46 10054.4 1824.40 10521.6 1825.70
#Mann=3,-1,0
  1801.3    0.05       0  4990.0    0.05       0  5017.0    0.05       0
Bank Sta=4990,5017
Exp/Cntr=0.3,0.1

Type RM Length L Ch R = 1,773852,2785,2785,2785
BEGIN DESCRIPTION:
Clear Fork Brazos Rv 178.0
END DESCRIPTION:
XS GIS Cut Line= 3
      1449704.97      6940237.96      1447705.00      6937238.00
      1442704.98      6932237.98
#Sta/Elev= 30
  1389.5 1831.52  1520.2 1830.97  1988.9 1820.63  2024.9 1816.59  2082.0 1813.55
  2118.1 1814.11  2226.2 1808.89  2370.5 1805.09  3467.2 1804.27  3697.0 1805.67
  4987.5 1795.20  4989.2 1788.35  4991.5 1787.35  5016.2 1788.35  5037.4 1790.62
  5051.6 1794.39  5178.9 1795.25  5277.8 1799.11  7936.6 1799.69  8403.3 1801.56
  8827.5 1808.65  9273.0 1811.74  9492.2 1814.88  9506.3 1816.55  9591.2 1814.71
  9718.5 1818.14 10708.4 1830.96 11443.8 1837.36 11838.8 1844.40 12066.1 1849.34
#Mann=4,-1,0
  1389.5    0.05       0  4989.2    0.05       0  5016.2    0.05       0
 11838.8    0.12       0
Bank Sta=4989.2,5016.2
Exp/Cntr=0.3,0.1

Type RM Length L Ch R = 1,771067,175,175,175
BEGIN DESCRIPTION:
Mapping XS 698f5e84
END DESCRIPTION:
XS GIS Cut Line= 4
      1451728.21      6939807.75      1450284.28      6935498.39
      1448742.09      6935057.77      1445168.08      6934320.95
#Sta/Elev= 30
  -981.3 1821.52  -570.3 1806.59  -140.1 1799.92  3320.6 1796.67  3363.6 1800.35
  3415.3 1797.34  3944.8 1795.76  4790.0 1796.76  4987.6 1792.39  4990.0 1785.05
  4993.0 1784.05  5026.0 1785.05  5050.0 1792.81  5542.5 1797.91  6022.1 1793.71
  8074.4 1799.93  8094.8 1804.26  8111.6 1801.86  8116.7 1805.01  8207.1 1801.00
  8212.2 1805.57  8257.4 1800.46  8262.5 1804.48  8307.6 1800.31  8312.8 1803.59
  8350.1 1802.58  8363.0 1806.71  8390.9 1803.00  8493.0 1803.39  8816.6 1808.69
#Mann=3,-1,0
  -981.3    0.05       0  4990.0   0.035       0  5026.0    0.05       0
Bank Sta=4990,5026
Exp/Cntr=0.3,0.1

Type RM Length L Ch R = 1,770892,1385,1385,1385
BEGIN DESCRIPTION:
Mapping XS d7e67f5c
END DESCRIPTION:
XS GIS Cut Line= 5
      1451804.85      6939851.58      1450224.96      6935218.77
      1448996.29      6934964.56      1448623.46      6934947.61
      1445335.74      6934024.00
#Sta/Elev= 30
 -1325.3 1821.64 -1119.9 1818.35  -848.4 1806.65  -415.0 1799.65  3058.0 1796.92
  3094.9 1800.39  3137.1 1797.42  3402.8 1798.25  3942.8 1795.15  4680.6 1796.15
  4822.3 1793.52  4945.6 1794.71  4978.0 1785.61  4981.0 1784.61  5014.0 1785.61
  5015.7 1793.90  5025.7 1794.87  5445.1 1792.19  5497.0 1796.70  5569.7 1797.11
  5736.6 1791.53  5756.7 1792.32  5777.5 1796.24  5912.1 1795.55  6098.1 1799.50
  6161.8 1797.14  6504.0 1796.08  7472.8 1798.20  7979.6 1800.75  8612.4 1808.20
#Mann=3,-1,0
 -1325.3    0.05       0  4978.0    0.03       0  5014.0    0.05       0
Bank Sta=4978,5014
Exp/Cntr=0.3,0.1

Type RM Length L Ch R = 1,769507,1719,1719,1719
BEGIN DESCRIPTION:
Mapping XS 289047ad
END DESCRIPTION:
XS GIS Cut Line= 6
      1451848.63      6939774.90      1450285.63      6935139.99
      1448849.85      6934503.68      1448050.38      6934095.79
      1447267.22      6934242.63      1445718.61      6933851.40
#Sta/Elev= 30
 -2567.4 1819.43 -2379.7 1815.24 -2322.0 1811.66 -2064.1 1804.42 -1692.5 1799.46
  1780.4 1796.55  1819.5 1800.14  1851.2 1797.43  1893.4 1796.89  2948.1 1795.88
  3560.6 1791.82  3877.8 1795.64  4667.5 1795.13  4756.4 1794.81  4832.0 1787.77
  4848.3 1789.94  4960.2 1793.54  4970.4 1792.92  4980.5 1789.64  4982.0 1787.05
  4985.0 1786.05  5018.0 1787.05  5021.2 1793.84  5031.4 1795.44  5052.5 1798.00
  5100.0 1799.42  5807.6 1796.99  6230.5 1797.63  6894.7 1801.75  7186.0 1806.39
#Mann=3,-1,0
 -2567.4    0.05       0  4982.0   0.035       0  5018.0    0.05       0
Bank Sta=4982,5018
Exp/Cntr=0.3,0.1

Type RM Length L Ch R = 1,767788,3218,3218,3218
BEGIN DESCRIPTION:
Mapping XS 7c27397e
END DESCRIPTION:
XS GIS Cut Line= 4
      1451980.00      6939884.39      1450305.94      6935089.91
      1448555.51      6934228.15      1447604.00      6932289.25
#Sta/Elev= 30
 -3187.7 1822.64 -3124.8 1822.29 -2850.6 1812.00 -2534.8 1803.64 -2250.7 1799.88
  1320.7 1796.55  1360.2 1800.21  1391.2 1797.14  1427.6 1796.81  2148.1 1796.88
  2205.0 1791.26  2227.4 1791.06  2266.8 1795.66  2384.7 1793.44  2401.6 1795.97
  2429.6 1796.34  3126.1 1791.87  3753.1 1795.30  4733.0 1795.26  4761.5 1792.79
  4955.8 1787.79  4978.1 1790.44  4982.0 1783.50  4985.0 1782.50  5018.0 1783.50
  5036.9 1785.96  5044.9 1791.36  5053.9 1792.08  5223.1 1797.03  6001.5 1801.36
#Mann=3,-1,0
 -3187.7    0.05       0  4982.0    0.05       0  5018.0    0.05       0
Bank Sta=4982,5018
Exp/Cntr=0.3,0.1

Type RM Length L Ch R = 1,764570,2737,2737,2737
BEGIN DESCRIPTION:
Mapping XS 25627341
END DESCRIPTION:
XS GIS Cut Line= 4
      1452316.96      6940280.57      1450198.91      6934534.04
      1449365.58      6932450.71      1447889.94      6931773.65
#Sta/Elev= 30
  -841.8 1830.28  -331.5 1819.61   -37.7 1818.17    56.2 1810.98   189.9 1805.06
   453.2 1799.97  4159.4 1796.38  4202.0 1800.15  4223.3 1797.48  4372.5 1796.02
  4876.7 1796.50  4948.0 1791.63  4962.7 1788.72  4980.5 1780.33  4982.8 1779.33
  5007.5 1780.33  5012.0 1789.48  5214.5 1786.95  5251.2 1788.22  5289.1 1794.28
  5321.5 1791.43  7507.8 1792.14  7525.2 1794.94  7544.3 1792.87  7549.8 1795.37
  7567.3 1793.24  8176.2 1795.30  8410.5 1801.93  8697.4 1800.52  9150.0 1803.25
#Mann=3,-1,0
  -841.8    0.05       0  4980.5    0.04       0  5007.5    0.05       0
Bank Sta=4980.5,5007.5
Exp/Cntr=0.3,0.1

Type RM Length L Ch R = 1,761833,9262,9262,9262
BEGIN DESCRIPTION:
Mapping XS d492d32d
END DESCRIPTION:
XS GIS Cut Line= 4
      1454695.44      6939950.72      1451500.99      6932815.29
      1450077.38      6931617.38      1449955.85      6929568.79
#Sta/Elev= 30
 -3614.3 1820.08 -3083.5 1808.99 -2863.8 1803.40 -2833.4 1800.76 -2636.2 1798.13
   738.4 1796.96   783.7 1795.21  3593.3 1790.27  3986.3 1790.04  4047.2 1791.93
  4159.6 1789.66  4681.9 1791.29  4908.3 1785.48  4986.4 1786.71  4993.0 1777.53
  4995.3 1776.53  5020.0 1777.53  5043.6 1787.86  5086.5 1791.64  5253.0 1789.76
  5320.6 1788.84  5370.0 1784.94  5405.1 1789.78  5444.9 1790.71  5610.6 1788.92
  5781.0 1796.17  5852.5 1803.78  5887.7 1804.76  7375.8 1807.78  8116.3 1815.95
#Mann=5,-1,0
 -3614.3    0.05       0  4993.0    0.05       0  5020.0    0.05       0
  5253.0    0.12       0  5444.9    0.05       0
Bank Sta=4993,5020
Exp/Cntr=0.3,0.1

Type RM Length L Ch R = 1,752571,2450,2450,2450
BEGIN DESCRIPTION:
Mapping XS 3b9d22b6
END DESCRIPTION:
XS GIS Cut Line= 3
      1458028.79      6937988.93      1454712.80      6932225.01
      1452021.86      6929846.57
#Sta/Elev= 30
 -3133.7 1838.98 -2960.5 1832.46 -2901.9 1833.08 -2874.2 1829.90 -2279.3 1808.16
 -2025.1 1804.96 -2002.0 1800.69 -1152.5 1795.48   779.2 1792.51   816.6 1795.32
   838.1 1792.78  1234.8 1790.81  3021.3 1787.28  3654.1 1789.12  4901.1 1787.46
  4964.9 1780.14  4986.5 1773.99  4988.8 1772.99  5013.5 1773.99  5014.2 1778.82
  5021.2 1779.35  5056.9 1780.24  5077.8 1777.07  5128.0 1778.51  5191.6 1782.99
  5226.7 1788.56  6069.9 1790.97  6402.8 1801.21  6799.3 1808.31  7107.4 1810.61
#Mann=3,-1,0
 -3133.7    0.05       0  4986.5    0.05       0  5013.5    0.05       0
Bank Sta=4986.5,5013.5
Exp/Cntr=0.3,0.1

Type RM Length L Ch R = 1,750121,2580,2580,2580
BEGIN DESCRIPTION:
Clear Fork Brazos Rv 174.0
END DESCRIPTION:
XS GIS Cut Line= 3
      1458370.32      6937650.89      1455389.68      6930412.19
      1455300.97      6928708.94
#Sta/Elev= 30
 -3202.7 1823.49 -2853.5 1815.98 -2799.4 1818.19 -2734.6 1813.04 -1988.3 1795.72
 -1626.0 1794.68 -1588.2 1798.05 -1543.4 1793.67 -1471.5 1793.18   412.5 1791.29
   434.1 1789.40   473.5 1791.40  2258.7 1785.97  3729.5 1787.11  4740.0 1785.18
  4808.4 1779.05  4840.1 1778.54  4860.2 1774.77  4900.2 1778.58  4980.3 1778.50
  4990.3 1777.26  4992.6 1771.19  4994.9 1770.19  5019.6 1771.19  5040.4 1779.95
  5110.5 1791.55  5280.7 1798.84  5380.9 1801.72  6061.8 1808.17  6331.2 1813.99
#Mann=3,-1,0
 -3202.7    0.05       0  4992.6    0.05       0  5019.6    0.05       0
Bank Sta=4992.6,5019.6
Exp/Cntr=0.3,0.1

Type RM Length L Ch R = 1,747541,1244,1244,1244
BEGIN DESCRIPTION:
Clear Fork Brazos Rv 173.0
END DESCRIPTION:
XS GIS Cut Line= 3
      1461504.97      6934337.97      1457505.00      6929338.00
      1456004.97      6928337.98
#Sta/Elev= 30
 -1402.6 1806.46 -1352.2 1806.48 -1325.0 1801.15 -1296.2 1799.55 -1032.1 1797.75
  -976.0 1794.09  -912.0 1793.11  -840.0 1795.13  -698.3 1792.70  -627.1 1794.23
  -300.5 1789.95   226.2 1786.69  1286.7 1786.22  1899.0 1782.28  3136.4 1778.49
  3491.7 1781.81  4872.4 1783.31  4964.5 1773.78  4980.2 1769.45  4982.4 1768.45
  5007.2 1769.45  5008.0 1773.10  5014.0 1776.11  5059.1 1776.74  5101.1 1783.65
  5281.4 1784.18  5433.2 1791.46  5590.9 1795.26  6465.2 1803.73  6803.3 1815.99
#Mann=3,-1,0
 -1402.6    0.05       0  4980.2    0.05       0  5007.2    0.05       0
Bank Sta=4980.2,5007.2
Exp/Cntr=0.3,0.1

Type RM Length L Ch R = 1,746297,6425,6425,6425
BEGIN DESCRIPTION:
Mapping XS 99c61be0
END DESCRIPTION:
XS GIS Cut Line= 3
      1462283.45      6933652.62      1459800.79      6930041.48
      1457231.37      6927524.14
#Sta/Elev= 30
 -1165.3 1795.40  -926.4 1795.11  -710.7 1790.89  -370.9 1788.50  -335.1 1789.46
  -329.0 1791.78  -293.2 1789.15    53.3 1785.28   648.5 1783.50  1116.7 1779.41
  1576.8 1782.20  2784.3 1777.49  3130.1 1779.83  3251.8 1779.45  3393.1 1775.39
  3534.6 1779.80  4227.6 1782.43  4354.9 1780.23  4899.4 1782.55  4920.6 1784.25
  4970.2 1773.88  4983.9 1767.67  4986.1 1766.27  5010.9 1767.67  5012.6 1776.06
  5111.6 1774.04  5154.0 1781.46  5840.0 1783.45  6165.1 1790.66  6814.0 1792.14
#Mann=3,-1,0
 -1165.3    0.05       0  4983.9   0.035       0  5010.9    0.05       0
Bank Sta=4983.9,5010.9
Exp/Cntr=0.3,0.1

Type RM Length L Ch R = 1,739872,2308,2308,2308
BEGIN DESCRIPTION:
Mapping XS 7518104d
END DESCRIPTION:
XS GIS Cut Line= 3
      1463325.08      6932680.34      1460495.23      6927454.68
      1457856.35      6925388.71
#Sta/Elev= 30
  -982.6 1790.95  1112.6 1776.98  4524.2 1779.16  4802.9 1777.64  4841.0 1772.16
  4868.6 1771.38  4890.4 1766.93  4979.2 1771.18  4985.8 1769.83  4988.0 1764.73
  4990.3 1763.83  5015.0 1764.73  5049.8 1778.93  5072.4 1779.68  5805.7 1779.73
  5919.6 1776.19  5940.4 1770.58  5990.1 1775.14  6083.2 1777.99  6182.7 1778.08
  6360.8 1772.92  6382.8 1779.61  6574.2 1777.52  6810.2 1780.53  6909.7 1774.88
  6924.1 1779.07  7017.2 1784.38  7137.5 1781.09  7522.7 1787.50  8311.5 1791.19
#Mann=3,-1,0
  -982.6    0.05       0  4988.0    0.05       0  5015.0    0.05       0
Bank Sta=4988,5015
Exp/Cntr=0.3,0.1

Type RM Length L Ch R = 1,737564,1593,1593,1593
BEGIN DESCRIPTION:
Mapping XS ab1d7112
END DESCRIPTION:
XS GIS Cut Line= 3
      1463584.33      6931895.16      1461969.74      6926877.79
      1457056.57      6923127.81
#Sta/Elev= 30
  -661.8 1784.63  1026.5 1775.58  1799.7 1774.58  2381.7 1776.63  4712.5 1776.25
  4783.2 1778.08  4804.0 1777.07  4868.4 1765.51  4891.2 1766.15  4904.3 1768.43
  4952.4 1768.78  4961.9 1767.80  4965.9 1765.71  4976.5 1762.62  4978.7 1761.72
  5003.5 1762.62  5004.9 1770.29  5011.8 1773.00  5040.9 1777.02  5269.1 1779.62
  5924.2 1780.41  6102.9 1782.26  6853.1 1779.91  6973.7 1781.90  7258.5 1781.66
  7416.4 1785.28  8029.5 1785.10  8314.3 1787.99  9684.6 1791.50 10789.7 1799.57
#Mann=5,-1,0
  -661.8    0.05       0  4952.4    0.12       0  4965.9    0.05       0
  4976.5    0.05       0  5003.5    0.05       0
Bank Sta=4976.5,5003.5
Exp/Cntr=0.3,0.1

Type RM Length L Ch R = 1,735971,3296,3296,3296
BEGIN DESCRIPTION:
Mapping XS de2d1ca5
END DESCRIPTION:
XS GIS Cut Line= 4
      1463485.04      6930832.65      1463827.67      6929478.44
      1462506.10      6924991.62      1460478.43      6923970.62
#Sta/Elev= 30
  -553.9 1780.15    -5.6 1782.29   895.6 1775.65  2746.0 1771.36  3492.9 1775.89
  4555.4 1774.88  4773.6 1766.66  4976.3 1767.89  4992.5 1767.28  4994.0 1760.63
  4997.0 1759.63  5030.0 1760.63  5055.0 1767.22  5086.7 1768.34  5114.8 1762.50
  5120.0 1766.97  5138.4 1761.90  5201.0 1762.42  5220.0 1766.95  5232.3 1761.61
  5258.6 1767.25  5263.8 1762.42  5291.9 1772.71  5297.1 1768.87  5315.7 1774.47
  6095.3 1775.61  6220.5 1774.79  6269.7 1770.64  6359.0 1775.24  7790.6 1784.39
#Mann=5,-1,0
  -553.9    0.05       0  4994.0    0.05       0  5030.0    0.05       0
  6095.3    0.12       0  6220.5    0.05       0
Bank Sta=4994,5030
Exp/Cntr=0.3,0.1

Type RM Length L Ch R = 1,732675,481,481,481
BEGIN DESCRIPTION:
Clear Fork Brazos Rv 169.0
END DESCRIPTION:
XS GIS Cut Line= 3
      1463636.41      6931113.88      1464680.66      6926169.23
      1465580.42      6922157.50
#Sta/Elev= 30
   -57.7 1781.86   714.9 1781.94  1651.8 1775.19  4077.9 1772.85  4311.3 1770.13
  4394.3 1773.25  4833.7 1773.68  4925.7 1763.63  4966.6 1763.62  4988.8 1757.43
  4991.0 1756.43  5015.8 1757.43  5035.9 1762.47  5041.0 1758.54  5058.8 1763.70
  5132.9 1763.02  5171.1 1767.46  5224.7 1766.49  5284.2 1771.98  5408.3 1772.67
  5786.4 1768.95  5929.9 1774.14  7538.9 1773.85  7702.9 1773.28  7736.7 1767.28
  7780.0 1773.33  7948.8 1776.74  8509.4 1783.14  8574.0 1786.94  9107.4 1793.88
#Mann=3,-1,0
   -57.7    0.05       0  4988.8    0.05       0  5015.8    0.05       0
Bank Sta=4988.8,5015.8
Exp/Cntr=0.3,0.1

Type RM Length L Ch R = 1,732194,3131,3131,3131
BEGIN DESCRIPTION:
Clear Fork Brazos Rv 168.0
END DESCRIPTION:
XS GIS Cut Line= 3
      1464244.05      6930801.39      1465094.74      6926218.07
      1466188.26      6922382.08
#Sta/Elev= 30
   269.0 1783.14   892.9 1782.52  1513.3 1776.22  4584.9 1773.22  4706.9 1772.31
  4741.4 1771.27  4778.1 1766.03  4904.9 1765.54  4948.0 1761.08  4982.7 1761.70
  4989.6 1758.19  4991.1 1757.19  5007.6 1758.19  5013.9 1763.99  5083.7 1765.92
  5244.7 1772.66  6517.4 1772.90  6886.9 1768.93  7105.5 1769.55  7139.4 1767.31
  7173.2 1768.90  7207.0 1768.00  7218.3 1763.29  7246.1 1762.34  7251.3 1766.90
  7397.0 1772.77  7551.1 1772.16  8164.8 1783.85  8523.9 1787.92  8919.4 1798.62
#Mann=5,-1,0
   269.0    0.05       0  4982.7    0.12       0  4989.6    0.07       0
  5007.6    0.12       0  5083.7    0.05       0
Bank Sta=4989.6,5007.6
Exp/Cntr=0.3,0.1

Type RM Length L Ch R = 1,729063,1244,1244,1244
BEGIN DESCRIPTION:
Clear Fork Brazos Rv 167.0
END DESCRIPTION:
XS GIS Cut Line= 3
      1466955.00      6928787.98      1467046.44      6924741.61
      1467189.11      6922601.57
#Sta/Elev= 30
   661.5 1800.94   879.7 1799.40   971.6 1796.81  1001.6 1798.85  1051.6 1795.98
  1271.6 1789.96  1631.7 1786.71  2081.8 1774.13  2461.9 1772.04  3292.2 1773.20
  3612.2 1768.51  4512.5 1771.15  4612.5 1768.66  4742.6 1768.81  4832.8 1762.66
  4882.9 1761.11  4953.1 1763.16  4973.1 1761.99  4984.4 1758.29  4986.7 1757.29
  5011.4 1758.29  5013.2 1760.67  5043.3 1768.51  5113.4 1771.48  5153.5 1770.26
  5173.5 1772.84  5516.7 1778.52  5962.7 1782.19  6065.5 1781.47  6853.7 1792.05
#Mann=3,-1,0
   661.5    0.05       0  4984.4    0.05       0  5011.4    0.05       0
Bank Sta=4984.4,5011.4
Exp/Cntr=0.3,0.1

Type RM Length L Ch R = 1,727819,1659,1659,1659
BEGIN DESCRIPTION:
Mapping XS c1ba433a
END DESCRIPTION:
XS GIS Cut Line= 3
      1467482.39      6927536.84      1467873.97      6924991.62
      1467776.07      6923457.91
#Sta/Elev= 30
  2722.6 1778.41  3308.3 1772.48  4077.2 1773.59  4117.7 1771.67  4866.4 1770.11
  4937.2 1766.47  4947.6 1762.33  4957.4 1754.16  4966.0 1752.05  4969.0 1751.05
  5002.0 1752.05  5005.8 1763.25  5119.3 1762.30  5137.3 1760.72  5142.4 1758.37
  5210.7 1760.75  5230.6 1758.31  5268.9 1767.29  5273.9 1765.56  5291.3 1768.75
  5481.8 1770.65  5702.2 1768.26  5782.4 1770.13  5882.6 1777.06  5962.7 1788.60
  6153.1 1788.25  6173.2 1785.89  6604.0 1782.83  6724.3 1786.90  6834.6 1787.73
#Mann=3,-1,0
  2722.6    0.05       0  4966.0    0.05       0  5002.0    0.05       0
Bank Sta=4966,5002
Exp/Cntr=0.3,0.1

Type RM Length L Ch R = 1,726160,5220,5220,5220
BEGIN DESCRIPTION:
Clear Fork Brazos Rv 166.0
END DESCRIPTION:
XS GIS Cut Line= 3
      1469673.74      6928479.40      1469205.00      6924638.00
      1469205.00      6923137.99
#Sta/Elev= 30
  1121.0 1794.28  1243.3 1793.79  1283.6 1796.68  1334.0 1791.83  1716.8 1778.67
  1988.8 1771.81  2895.5 1771.43  3464.1 1768.98  3661.1 1766.14  3842.4 1768.93
  4416.7 1770.89  4567.8 1764.68  4678.6 1764.64  4859.9 1760.02  4980.8 1760.94
  4988.4 1757.93  4989.8 1751.14  4992.0 1750.14  5016.8 1751.14  5050.9 1761.12
  5110.5 1760.38  5208.4 1760.74  5407.4 1763.36  5442.2 1764.10  5460.9 1766.66
  5470.9 1770.17  5510.9 1773.09  5730.9 1781.18  6140.9 1788.22  6490.9 1790.25
#Mann=7,-1,0
  1121.0    0.05       0  4989.8    0.05       0  5016.8    0.05       0
  5110.5    0.12       0  5208.4    0.05       0  5407.4    0.12       0
  5442.2    0.05       0
Bank Sta=4989.8,5016.8
Exp/Cntr=0.3,0.1

Type RM Length L Ch R = 1,720940,3866,3866,3866
BEGIN DESCRIPTION:
Clear Fork Brazos Rv 165.0
END DESCRIPTION:
XS GIS Cut Line= 3
      1470741.46      6928062.74      1470559.15      6927307.48
      1470705.00      6922238.02
#Sta/Elev= 30
  4261.1 1789.95  4824.0 1774.18  4860.7 1770.07  4865.9 1771.96  4883.2 1764.91
  4902.6 1763.46  4907.7 1767.29  4944.5 1755.97  4986.1 1754.64  4988.5 1749.98
  4990.7 1748.98  5015.5 1749.98  5027.2 1752.70  5033.4 1757.78  5117.6 1753.03
  5157.6 1758.42  5317.6 1764.51  5987.9 1763.27  6106.8 1766.90  6288.0 1767.04
  6460.8 1763.27  6608.2 1769.73  8398.9 1770.91  9009.2 1781.94  9219.3 1787.11
  9237.3 1790.48  9299.3 1792.76  9459.4 1794.31  9779.5 1805.31 10109.6 1812.06
#Mann=3,-1,0
  4261.1     0.1       0  4988.5    0.05       0  5015.5     0.1       0
Bank Sta=4988.5,5015.5
Exp/Cntr=0.3,0.1

Type RM Length L Ch R = 1,717074,3105,3105,3105
BEGIN DESCRIPTION:
Clear Fork Brazos Rv 164.0
END DESCRIPTION:
XS GIS Cut Line= 3
      1472455.00      6928637.97      1472512.20      6925496.21
      1471991.44      6922593.94
#Sta/Elev= 30
  1851.2 1802.14  2641.3 1778.36  2675.7 1782.64  3411.4 1760.67  3991.5 1766.86
  4481.6 1764.76  4591.6 1757.28  4891.7 1752.67  4961.7 1754.97  4971.7 1752.10
  4983.5 1743.83  4985.8 1742.83  5010.5 1743.83  5012.0 1750.21  5032.3 1755.81
  5133.9 1758.49  5172.6 1753.34  5194.9 1757.99  5250.6 1760.91  5337.1 1765.35
  5402.7 1763.98  5456.4 1768.40  5672.4 1771.48  5852.7 1780.60  6254.1 1778.99
  6718.8 1793.24  7237.0 1797.35  7609.2 1788.84  7866.9 1790.55  7942.1 1794.64
#Mann=4,-1,0
  1851.2     0.1       0  4983.5    0.05       0  5010.5    0.07       0
  5250.6    0.07       0
Bank Sta=4983.5,5010.5
Exp/Cntr=0.3,0.1

Type RM Length L Ch R = 1,713969,1266,1266,1266
BEGIN DESCRIPTION:
Mapping XS 6079fd2c
END DESCRIPTION:
XS GIS Cut Line= 4
      1472817.63      6928466.86      1473013.41      6927602.13
      1473894.46      6926525.30      1476129.71      6924436.89
#Sta/Elev= 30
  3647.7 1789.75  4160.4 1781.22  4198.5 1786.48  4515.9 1784.78  4837.7 1773.53
  4915.0 1768.58  4959.3 1755.12  4986.1 1754.14  4992.0 1741.65  4995.0 1740.65
  5028.0 1741.65  5048.0 1750.26  5064.4 1754.48  5121.1 1754.46  5134.7 1750.74
  5163.4 1755.10  5299.1 1756.55  5383.8 1765.30  5412.5 1762.75  5482.9 1768.32
  7109.1 1767.05  7205.5 1766.97  8421.6 1767.79  8524.2 1763.73  8539.1 1763.38
  8690.8 1767.59  8737.7 1769.01  8830.0 1773.17  8877.0 1780.27  8984.7 1784.57
#Mann=15,-1,0
  3647.7     0.1       0  4837.7    0.12       0  4915.0     0.1       0
  4959.3    0.12       0  4992.0    0.05       0  5028.0    0.12       0
  5048.0     0.1       0  7109.1    0.12       0  7205.5    0.05       0
  8524.2    0.12       0  8539.1    0.05       0  8690.8    0.12       0
  8737.7    0.05       0  8830.0    0.12       0  8877.0    0.05       0
#XS Ineff=2,0
       0                 6200.00    0.00 1779.35
Permanent Ineff=
       F       F
Bank Sta=4992,5028
Exp/Cntr=0.3,0.1

Type RM Length L Ch R = 1,712703,1307,1307,1307
BEGIN DESCRIPTION:
Clear Fork Brazos Rv 163.0
END DESCRIPTION:
XS GIS Cut Line= 3
      1473155.02      6928537.99      1474155.00      6928038.00
      1477654.97      6926038.02
#Sta/Elev= 30
  3869.7 1786.73  4017.8 1784.51  4070.9 1788.53  4392.4 1767.67  4487.4 1769.02
  4576.8 1766.42  4607.6 1758.37  4697.0 1751.34  4800.4 1753.38  4808.8 1751.30
  4951.4 1755.72  4979.3 1752.01  4984.9 1746.41  4986.9 1738.96  4989.2 1737.86
  5013.9 1738.96  5017.2 1743.26  5033.1 1751.08  5045.3 1760.93  5060.4 1765.79
  6871.5 1761.96  7406.4 1764.56  7876.4 1759.40  8102.5 1762.82  8270.2 1761.11
  8484.0 1766.19  8682.7 1767.46  8747.5 1773.53  8806.5 1787.18  9018.8 1793.64
#Mann=3,-1,0
  3869.7     0.1       0  4986.9    0.05       0  5013.9     0.1       0
#XS Ineff=2,0
       0                 6200.00    0.00 1780.15
Permanent Ineff=
       F       F
Bank Sta=4986.9,5013.9
Exp/Cntr=0.3,0.1

Type RM Length L Ch R = 1,711396,1039,1039,1039
BEGIN DESCRIPTION:
Mapping XS d30e98d7
END DESCRIPTION:
XS GIS Cut Line= 3
      1473829.21      6930196.33      1474906.04      6928907.39
      1477679.73      6926655.80
#Sta/Elev= 30
  3270.0 1792.10  3550.0 1780.23  3663.2 1774.01  3734.8 1767.01  3827.2 1762.86
  4877.4 1763.56  4920.4 1760.97  4942.5 1755.96  4990.8 1750.64  4998.0 1740.25
  5001.0 1739.25  5034.0 1740.25  5040.3 1745.78  5054.7 1749.11  5085.7 1751.49
  5112.2 1750.20  5126.6 1751.67  5141.0 1753.81  5168.2 1762.33  5197.0 1764.63
  5304.0 1761.67  5609.3 1762.98  7046.1 1759.58  7124.4 1761.18  7357.8 1756.48
  7592.7 1762.35  7941.2 1763.19  8208.6 1766.25  8290.8 1767.85  8522.1 1772.00
#Mann=7,-1,0
  3270.0     0.1       0  4942.5    0.12       0  4998.0    0.05       0
  5034.0    0.12       0  5085.7     0.1       0  8208.6    0.12       0
  8290.8    0.05       0
#XS Ineff=2,0
    0.00 3153.10 1781.49 6200.00    0.00 1781.49
Permanent Ineff=
       F       F
Bank Sta=4998,5034
Exp/Cntr=0.3,0.1

Type RM Length L Ch R = 1,710357,1453,1453,1453
BEGIN DESCRIPTION:
Mapping XS ed52b66a
END DESCRIPTION:
XS GIS Cut Line= 3
      1474857.07      6931387.42      1476064.45      6928842.13
      1478267.04      6927226.90
#Sta/Elev= 30
  2712.1 1796.66  2820.3 1793.12  3054.6 1784.92  3331.3 1762.76  3430.9 1759.77
  4836.5 1763.13  4893.1 1760.38  4910.3 1754.82  4933.1 1751.05  4978.5 1750.80
  4984.1 1749.44  4987.5 1739.20  4991.3 1738.20  5032.5 1739.20  5035.7 1747.91
  5057.9 1757.47  5080.5 1761.78  5126.0 1763.03  5313.4 1759.50  5661.6 1761.87
  6261.6 1761.75  6391.0 1759.78  6520.6 1751.79  6541.5 1756.37  6641.8 1759.94
  6956.0 1764.16  7335.7 1763.46  7778.7 1765.93  8065.1 1771.23  8260.6 1778.61
#Mann=4,-1,0
  2712.1    0.12       0  2820.3     0.1       0  4987.5    0.05       0
  5032.5     0.1       0
#XS Ineff=2,0
       0                 6098.60    0.00 1778.80
Permanent Ineff=
       F       F
Bank Sta=4987.5,5032.5
Exp/Cntr=0.3,0.1

Type RM Length L Ch R = 1,708904,3968,3968,3968
BEGIN DESCRIPTION:
Clear Fork Brazos Rv 162.0
END DESCRIPTION:
XS GIS Cut Line= 3
      1475220.63      6932645.99      1477155.00      6929688.00
      1478655.00      6927188.00
#Sta/Elev= 30
  1477.5 1798.48  1753.1 1797.90  2317.1 1772.43  2410.6 1772.42  2461.9 1775.84
  2591.6 1763.96  2736.4 1757.58  4737.0 1761.53  4817.3 1758.59  4859.5 1752.44
  4931.9 1751.93  4953.0 1749.10  4962.1 1743.89  4968.1 1744.85  4976.0 1739.86
  4987.8 1738.79  4990.0 1737.69  5014.8 1738.79  5019.6 1748.08  5025.4 1749.27
  5136.2 1756.58  5252.8 1756.89  5295.6 1760.27  5421.5 1759.68  6652.3 1764.12
  7505.5 1772.57  7694.1 1777.97  7802.9 1786.68  7834.0 1792.19  7927.3 1796.38
#Mann=4,-1,0
  1477.5     0.1       0  4987.8    0.05       0  5014.8     0.1       0
  5421.5    0.05       0
#XS Ineff=2,0
       0                 5881.20    0.00 1782.29
Permanent Ineff=
       F       F
Bank Sta=4987.8,5014.8
Exp/Cntr=0.3,0.1

Type RM Length L Ch R = 1,704936,3449,3449,3449
BEGIN DESCRIPTION:
Clear Fork Brazos Rv 161.0
END DESCRIPTION:
XS GIS Cut Line= 3
      1478762.28      6935224.14      1479155.00      6931388.00
      1479309.16      6929338.68
#Sta/Elev= 30
  1149.0 1786.94  1421.4 1781.29  1698.0 1768.51  1714.4 1768.17  1728.2 1770.81
  1748.3 1768.00  1798.5 1766.46  1813.8 1763.58  1838.7 1765.57  2130.2 1761.36
  2582.6 1761.41  3175.7 1752.95  4552.8 1756.01  4743.8 1759.14  4784.0 1755.55
  4814.2 1747.68  4844.4 1744.54  4904.7 1748.76  4944.9 1748.42  4958.0 1747.03
  4982.0 1734.59  4984.3 1733.39  5009.0 1734.59  5015.2 1747.31  5025.2 1754.06
  5055.3 1758.56  5546.7 1755.76  5740.3 1757.19  6068.2 1765.13  7060.3 1764.63
#Mann=3,-1,0
  1149.0     0.1       0  4982.0    0.05       0  5009.0     0.1       0
Bank Sta=4982,5009
Exp/Cntr=0.3,0.1

Type RM Length L Ch R = 1,701487,6005,6005,6005
BEGIN DESCRIPTION:
Clear Fork Brazos Rv 160.0
END DESCRIPTION:
XS GIS Cut Line= 3
      1481184.15      6937125.22      1482155.00      6932688.00
      1481355.00      6928588.01
#Sta/Elev= 30
   457.9 1796.88   946.4 1785.73  1050.3 1774.27  1187.0 1769.78  1563.5 1767.48
  1714.1 1758.73  2213.5 1751.11  3802.2 1748.07  4833.8 1753.52  4938.4 1748.16
  4969.4 1746.30  4985.8 1733.52  4988.0 1732.32  5012.8 1733.52  5020.5 1735.37
  5025.9 1743.87  5083.7 1746.49  5232.2 1745.16  5500.3 1751.38  6986.9 1747.03
  7320.9 1757.52  8270.6 1764.36  8617.0 1773.09  8733.9 1770.38  8810.6 1771.84
  8888.6 1781.08  8922.7 1789.08  8953.3 1802.38  8991.8 1806.52  9177.4 1809.99
#Mann=5,-1,0
   457.9     0.1       0  4938.4     0.1       0  4985.8    0.05       0
  5012.8     0.1       0  5083.7     0.1       0
Bank Sta=4985.8,5012.8
Exp/Cntr=0.3,0.1

Type RM Length L Ch R = 1,695482,477,477,477
BEGIN DESCRIPTION:
Mapping XS f4c9daf9
END DESCRIPTION:
XS GIS Cut Line= 2
      1483088.56      6937458.10      1484876.39      6929751.35
#Sta/Elev= 30
  -540.4 1783.91  -427.4 1784.44  -225.7 1779.68   -98.9 1781.08   250.1 1769.22
   630.0 1763.65   658.2 1764.72   748.6 1761.88   972.2 1760.89  1190.6 1751.35
  1451.2 1748.98  1770.8 1748.33  2079.7 1750.55  2796.0 1746.58  4786.7 1748.72
  4821.9 1748.81  4949.9 1739.25  4972.3 1739.37  4982.6 1735.87  4986.5 1727.63
  4988.8 1726.43  5013.5 1727.63  5033.9 1737.93  5040.3 1739.31  5045.5 1737.96
  5071.0 1742.47  5116.0 1747.78  5167.3 1748.69  6645.6 1747.84  7371.0 1752.08
#Mann=5,-1,0
  -540.4     0.1       0  4786.7     0.1       0  4986.5    0.05       0
  5013.5     0.1       0  5071.0     0.1       0
Bank Sta=4986.5,5013.5
Exp/Cntr=0.3,0.1

Type RM Length L Ch R = 1,695005,1458,1458,1458
BEGIN DESCRIPTION:
Mapping XS 9c229a51
END DESCRIPTION:
XS GIS Cut Line= 2
      1483487.87      6937527.55      1485310.80      6929819.17
#Sta/Elev= 30
  -692.3 1787.74  -528.3 1781.71  -374.0 1781.91  -343.4 1772.80  -331.7 1772.28
  -271.5 1774.47  -115.2 1772.32   -78.0 1777.09    11.7 1770.21   119.0 1779.95
   180.7 1768.94   283.4 1768.45   375.9 1761.57   468.4 1761.39   499.2 1769.06
   519.8 1769.94   540.3 1760.47   560.9 1758.31   967.5 1749.50  2092.0 1745.55
  4856.2 1747.36  4887.0 1739.03  4970.0 1737.38  4980.5 1727.79  4982.8 1726.59
  5007.5 1727.79  5020.6 1741.10  5102.8 1747.05  6448.9 1745.90  7228.7 1751.17
#Mann=3,-1,0
  -692.3    0.05       0  4980.5   0.035       0  5007.5    0.05       0
Bank Sta=4980.5,5007.5
Exp/Cntr=0.3,0.1

Type RM Length L Ch R = 1,693547,5790,5790,5790
BEGIN DESCRIPTION:
Clear Fork Brazos Rv 159.0
END DESCRIPTION:
XS GIS Cut Line= 3
      1486704.98      6936734.55      1486205.00      6931888.00
      1485715.58      6927361.25
#Sta/Elev= 30
   125.6 1778.71   665.7 1773.70   858.7 1767.78  1117.4 1756.50  1328.5 1751.06
  1750.7 1744.30  2896.8 1745.00  3580.1 1743.12  3691.0 1741.37  4851.9 1746.00
  4897.3 1745.50  4951.2 1741.34  4957.7 1740.79  4967.7 1735.92  4977.8 1728.72
  4982.8 1727.15  4985.1 1725.95  5009.8 1727.15  5018.0 1740.42  5049.9 1741.78
  5128.6 1740.40  5339.8 1746.23  5696.3 1743.45  6812.7 1742.65  7240.9 1748.42
  8117.7 1752.51  8327.2 1758.65  8427.7 1759.02  8953.8 1753.39  9551.0 1750.17
#Mann=5,-1,0
   125.6    0.05       0  4951.2     0.1       0  4982.8    0.07       0
  5009.8     0.1       0  5049.9    0.05       0
Bank Sta=4982.8,5009.8
Exp/Cntr=0.3,0.1

Type RM Length L Ch R = 1,687757,3430,3430,3430
BEGIN DESCRIPTION:
Mapping XS f4ade710
END DESCRIPTION:
XS GIS Cut Line= 2
      1491314.37      6933974.17      1487329.98      6927463.73
#Sta/Elev= 30
  1333.8 1784.85  1622.4 1780.41  1818.5 1770.94  1839.8 1771.68  1897.8 1767.44
  1962.4 1772.44  2008.1 1765.03  2093.3 1762.60  2151.3 1758.17  2203.5 1757.95
  2232.1 1754.57  2313.7 1750.89  2915.5 1737.09  4893.4 1742.27  4960.4 1735.98
  4975.5 1729.72  4982.8 1721.87  4985.0 1720.67  5009.8 1721.87  5010.7 1732.73
  5018.4 1735.08  5069.3 1735.95  5127.9 1744.30  5163.1 1741.43  6101.0 1741.85
  7222.0 1736.71  7891.4 1740.65  8211.3 1745.17  8508.6 1752.27  8966.7 1751.61
#Mann=3,-1,0
  1333.8    0.05       0  4982.8    0.05       0  5009.8    0.05       0
Bank Sta=4982.8,5009.8
Exp/Cntr=0.3,0.1

Type RM Length L Ch R = 1,684327,5119,5119,5119
BEGIN DESCRIPTION:
Mapping XS 35d44dbe
END DESCRIPTION:
XS GIS Cut Line= 3
      1493319.55      6932229.32      1492850.82      6931526.23
      1488789.17      6923585.18
#Sta/Elev= 30
  3496.2 1772.79  3803.1 1771.62  4034.4 1767.37  4235.7 1754.50  4341.2 1753.10
  4395.4 1747.78  4449.4 1746.68  4516.0 1741.28  4627.1 1737.05  4732.4 1735.56
  4788.5 1739.67  4804.8 1739.11  4821.4 1734.35  4884.0 1734.61  4960.3 1734.07
  4975.0 1719.96  4978.0 1718.76  5011.0 1719.96  5013.2 1732.26  5049.1 1740.58
  5110.1 1737.38  5271.5 1736.70  8439.0 1733.98  8752.4 1735.88  8974.6 1732.50
  9324.3 1734.50  9657.5 1732.92 10201.6 1736.61 10662.4 1744.53 13260.7 1750.45
#Mann=4,-1,0
  3496.2    0.05       0  4884.0     0.1       0  4975.0    0.07       0
  5011.0    0.05       0
Bank Sta=4975,5011
Exp/Cntr=0.3,0.1

Type RM Length L Ch R = 1,679208,5036,5036,5036
BEGIN DESCRIPTION:
Clear Fork Brazos Rv 156.0
END DESCRIPTION:
XS GIS Cut Line= 3
      1494998.37      6931635.90      1494711.91      6929526.51
      1492654.61      6925047.33
#Sta/Elev= 30
   838.3 1763.07  1249.9 1762.13  1461.9 1745.48  1496.1 1739.41  1583.0 1738.66
  1633.4 1733.77  1683.9 1732.85  4215.9 1732.74  4479.8 1734.29  4577.2 1738.64
  4669.1 1733.13  4772.1 1736.25  4835.5 1730.27  4902.2 1728.44  4938.5 1731.31
  4956.0 1726.91  4959.5 1716.90  4963.2 1715.70  5004.5 1716.90  5007.4 1732.17
  5035.9 1735.76  5067.2 1732.88  5386.2 1730.18  5661.5 1729.45  5684.0 1732.48
  5716.5 1729.27  5873.4 1729.27  6252.1 1736.99  7049.1 1741.19  7896.1 1741.48
#Mann=3,-1,0
   838.3    0.05       0  4959.5    0.03       0  5004.5    0.05       0
Bank Sta=4959.5,5004.5
Exp/Cntr=0.3,0.1

Type RM Length L Ch R = 1,674172,5498,5498,5498
BEGIN DESCRIPTION:
Mapping XS 67d2fc04
END DESCRIPTION:
XS GIS Cut Line= 3
      1496430.66      6931401.49      1496378.57      6929943.17
      1494217.10      6922573.35
#Sta/Elev= 30
  4033.5 1757.99  4727.4 1751.72  4788.1 1747.50  4837.5 1744.58  4927.6 1729.21
  4984.1 1725.21  4987.6 1724.28  4988.8 1716.02  4992.6 1714.82  5033.8 1716.02
  5057.6 1728.20  5082.2 1727.35  5227.8 1727.34  5277.8 1731.89  5452.8 1732.01
  8544.9 1728.61  8853.8 1728.72  8885.0 1731.37  8978.8 1727.91  8999.7 1730.12
  9570.8 1727.06  9997.6 1735.45 10213.6 1736.18 10463.0 1735.58 10779.3 1727.77
 11062.1 1733.67 11100.7 1731.00 11156.9 1735.65 11566.1 1738.53 13173.0 1744.04
#Mann=6,-1,0
  4033.5    0.05       0  4788.1     0.1       0  4984.1    0.12       0
  4988.8    0.07       0  5033.8    0.12       0  5082.2    0.05       0
Bank Sta=4988.8,5033.8
Exp/Cntr=0.3,0.1

Type RM Length L Ch R = 1,668674,1008,1008,1008
BEGIN DESCRIPTION:
Mapping XS d4f81cd9
END DESCRIPTION:
XS GIS Cut Line= 3
      1498369.90      6931254.02      1498612.95      6926913.78
      1496911.56      6924049.19
#Sta/Elev= 30
  -943.2 1761.89  -696.8 1755.11  -346.2 1733.79   -35.8 1725.44  2578.3 1728.34
  3359.6 1724.82  3896.2 1726.62  3954.7 1727.81  3968.8 1731.69  4077.4 1726.30
  4646.3 1724.43  4720.3 1719.63  4771.4 1724.98  4960.0 1725.67  4991.2 1723.59
  4997.0 1721.38  4997.5 1712.47  5001.3 1711.47  5042.5 1712.47  5055.4 1723.49
  5108.1 1726.12  5363.3 1726.15  5390.5 1725.10  5399.4 1719.46  5457.6 1725.61
  5492.5 1722.60  5515.7 1727.13  5587.3 1723.10  5762.7 1728.12  6735.6 1733.80
#Mann=3,-1,0
  -943.2    0.05       0  4997.5   0.035       0  5042.5    0.05       0
Bank Sta=4997.5,5042.5
Exp/Cntr=0.3,0.1

Type RM Length L Ch R = 1,667666,4864,4864,4864
BEGIN DESCRIPTION:
Mapping XS 38bf1977
END DESCRIPTION:
XS GIS Cut Line= 3
      1498689.68      6931291.53      1499019.54      6926031.06
      1496432.74      6921204.68
#Sta/Elev= 30
 -1116.1 1764.38  -902.2 1761.61  -634.1 1739.58  -170.7 1724.69  2344.2 1727.79
  4487.0 1725.73  4678.7 1725.92  4728.2 1728.97  4759.5 1723.94  4929.7 1722.44
  4963.8 1718.06  4970.7 1710.92  4974.5 1709.72  5015.7 1710.92  5018.2 1721.20
  5023.9 1719.37  5062.1 1724.32  5587.6 1724.20  6606.2 1733.53  8276.3 1734.92
  8643.4 1739.38  8851.4 1748.41  8941.8 1748.08  9076.8 1748.74  9238.9 1754.24
  9275.9 1756.58  9360.7 1766.35  9426.5 1769.08  9536.1 1760.61  9630.6 1758.93
#Mann=7,-1,0
 -1116.1    0.05       0  4970.7    0.05       0  5015.7    0.05       0
  8941.8    0.12       0  9076.8    0.05       0  9238.9    0.12       0
  9275.9    0.05       0
Bank Sta=4970.7,5015.7
Exp/Cntr=0.3,0.1

Type RM Length L Ch R = 1,662802,4606,4606,4606
BEGIN DESCRIPTION:
Clear Fork Brazos Rv 154.0
END DESCRIPTION:
XS GIS Cut Line= 3
      1498855.00      6931988.00      1500355.00      6927488.00
      1503354.98      6922988.03
#Sta/Elev= 30
   255.6 1772.00   434.8 1766.41   614.0 1773.32   687.8 1766.97  1151.6 1753.96
  1446.7 1737.32  1900.0 1724.84  4735.5 1726.23  4819.8 1716.87  4977.9 1719.49
  4987.0 1705.74  4990.0 1704.54  5023.0 1705.74  5035.1 1717.01  5042.6 1719.24
  5093.7 1716.96  5222.9 1725.62  9044.7 1722.18  9073.3 1720.20  9095.8 1708.19
  9131.9 1716.64  9576.4 1719.64  9693.7 1720.02  9729.8 1731.14  9780.9 1761.65
  9807.5 1769.60 10003.2 1768.65 10270.6 1751.19 10348.8 1761.14 10407.3 1761.32
#Mann=5,-1,0
   255.6    0.05       0  4987.0    0.05       0  5023.0    0.05       0
  9576.4    0.12       0  9807.5    0.05       0
Bank Sta=4987,5023
Exp/Cntr=0.3,0.1

Type RM Length L Ch R = 1,658196,3659,3659,3659
BEGIN DESCRIPTION:
Clear Fork Brazos Rv 153.0
END DESCRIPTION:
XS GIS Cut Line= 3
      1501855.00      6932437.97      1502756.61      6927703.59
      1503355.00      6923438.03
#Sta/Elev= 30
   567.9 1761.63  1125.9 1748.13  1494.2 1749.93  1772.4 1744.72  1824.6 1748.99
  1881.8 1742.95  2491.8 1740.90  3373.3 1719.76  4558.3 1717.26  4935.0 1722.01
  4945.2 1719.52  4959.6 1703.85  4963.4 1702.65  5004.6 1703.85  5006.2 1714.32
  5036.8 1717.07  5372.7 1713.22  5557.7 1721.78  8634.4 1720.03  8684.9 1706.61
  8705.1 1713.97  8734.6 1717.26  8887.8 1718.65  8907.1 1718.99  9068.7 1725.42
  9152.9 1749.64  9179.7 1758.43  9331.2 1769.95  9523.1 1763.67  9694.7 1769.38
#Mann=7,-1,0
   567.9    0.05       0  4959.6    0.05       0  5004.6    0.05       0
  8734.6    0.12       0  8887.8     0.1       0  8907.1    0.12       0
  9152.9    0.05       0
Bank Sta=4959.6,5004.6
Exp/Cntr=0.3,0.1

Type RM Length L Ch R = 1,654537,2334,2334,2334
BEGIN DESCRIPTION:
Clear Fork Brazos Rv 152.0
END DESCRIPTION:
XS GIS Cut Line= 3
      1504178.94      6930328.36      1504655.00      6925488.00
      1504755.00      6924887.99
#Sta/Elev= 30
   143.9 1724.61   887.8 1729.18  1074.0 1727.81  1281.7 1720.89  1541.0 1718.19
  1561.1 1715.67  1731.9 1713.27  2092.2 1717.26  3120.6 1718.56  3520.5 1717.22
  3922.4 1718.76  4254.0 1712.28  4515.7 1715.01  4731.8 1713.79  4927.2 1713.11
  4947.3 1708.36  4956.2 1701.68  4960.0 1700.38  5001.2 1701.68  5005.1 1715.03
  5301.6 1713.67  5372.6 1717.63  5423.3 1729.06  5461.3 1733.81  5466.4 1729.26
  5494.2 1732.77  5527.2 1728.28  5575.3 1734.03  5588.0 1738.76  5615.9 1752.95
#Mann=5,-1,0
   143.9    0.05       0  4515.7    0.12       0  4731.8    0.05       0
  4956.2    0.04       0  5001.2    0.05       0
Bank Sta=4956.2,5001.2
Exp/Cntr=0.3,0.1

Type RM Length L Ch R = 1,652203,3380,3380,3380
BEGIN DESCRIPTION:
Clear Fork Brazos Rv 151.0
END DESCRIPTION:
XS GIS Cut Line= 3
      1505042.50      6930902.59      1506686.26      6925514.35
      1506809.04      6923871.52
#Sta/Elev= 30
  -566.9 1720.64   880.7 1726.80  1339.6 1714.74  1612.5 1711.84  2961.2 1716.46
  4322.1 1714.76  4324.3 1714.88  4425.8 1713.68  4527.2 1712.23  4740.2 1715.04
  4805.8 1708.07  4864.0 1710.76  4970.9 1710.37  4975.1 1708.71  4977.8 1700.29
  4980.8 1698.99  5013.8 1700.29  5020.9 1710.81  5046.0 1710.25  5062.0 1713.30
  5143.1 1713.96  5173.1 1709.34  5186.2 1710.73  5363.7 1718.96  5604.3 1723.94
  5724.7 1723.35  5915.2 1730.29  6105.7 1726.95  6165.9 1729.28  6713.9 1725.71
#Mann=9,-1,0
  -566.9    0.05       0  4322.1     0.1       0  4324.3    0.05       0
  4425.8     0.1       0  4527.2    0.05       0  4970.9     0.1       0
  4977.8    0.07       0  5013.8     0.1       0  5186.2    0.05       0
Bank Sta=4977.8,5013.8
Exp/Cntr=0.3,0.1
