HEC-RAS study Clear Fork Brazos Rv.prj: Clear Fork Brazos Rv Base Level Engineering

--- Clear Fork Brazos Rv.g01 (geometry) --- (continued)

Type RM Length L Ch R = 1,648823,5856,5856,5856
BEGIN DESCRIPTION:
Mapping XS 02894f41
END DESCRIPTION:
XS GIS Cut Line= 4
      1507380.32      6930594.31      1508040.03      6929170.72
      1508369.90      6927087.39      1508265.73      6923893.00
#Sta/Elev= 30
  1474.3 1721.93  2521.4 1721.51  3309.3 1708.32  4838.4 1714.97  4911.8 1707.44
  4969.7 1708.04  4979.9 1706.17  4982.0 1700.78  4985.0 1699.78  5018.0 1700.78
  5040.6 1708.21  5101.4 1705.57  5173.9 1710.62  6087.0 1713.03  6162.5 1712.18
  6232.6 1703.14  6306.8 1703.44  6368.4 1709.02  6372.2 1709.99  6377.2 1703.18
  6442.0 1712.03  6553.1 1713.23  6777.1 1711.69  6908.6 1709.77  7043.0 1708.60
  7053.0 1713.14  7193.8 1716.41  7623.3 1723.65  7663.3 1729.04  8348.7 1726.90
#Mann=13,-1,0
  1474.3    0.05       0  4911.8     0.1       0  4982.0    0.07       0
  5018.0     0.1       0  5173.9    0.05       0  6087.0     0.1       0
  6306.8    0.05       0  6368.4     0.1       0  6442.0    0.05       0
  6553.1    0.12       0  6777.1    0.05       0  6908.6    0.12       0
  7193.8    0.05       0
Bank Sta=4982,5018
Exp/Cntr=0.3,0.1

Type RM Length L Ch R = 1,642967,2547,2547,2547
BEGIN DESCRIPTION:
Clear Fork Brazos Rv 150.0
END DESCRIPTION:
XS GIS Cut Line= 3
      1507746.65      6933349.16      1510742.72      6926596.82
      1511623.76      6923701.17
#Sta/Elev= 30
 -2251.5 1728.50 -2162.7 1731.46 -2145.5 1729.61 -1647.3 1727.66  -962.9 1731.12
  -828.0 1730.21  -806.1 1726.29  -418.2 1719.95   112.8 1719.92  1007.9 1710.68
  2787.2 1708.46  4834.5 1711.56  4948.4 1711.31  4992.2 1703.34  4994.2 1693.33
  4997.2 1692.03  5030.2 1693.33  5035.9 1698.88  5053.7 1705.19  5076.9 1703.52
  5090.6 1698.95  5110.3 1702.69  5198.7 1702.58  5270.3 1709.63  6388.8 1711.81
  6629.2 1716.47  6669.0 1715.04  7155.1 1723.91  7636.0 1739.98  8162.4 1749.59
#Mann=5,-1,0
 -2251.5    0.05       0  4834.5     0.1       0  4994.2    0.07       0
  5030.2     0.1       0  5110.3    0.05       0
Bank Sta=4994.2,5030.2
Exp/Cntr=0.3,0.1

Type RM Length L Ch R = 1,640420,5743,5743,5743
BEGIN DESCRIPTION:
Mapping XS 115970a2
END DESCRIPTION:
XS GIS Cut Line= 5
      1512145.71      6932780.22      1512888.33      6928274.04
      1512786.90      6927194.26      1511918.84      6925753.29
      1511849.40      6923947.75
#Sta/Elev= 30
  -356.1 1720.39   801.5 1710.03  1845.4 1708.00  2193.4 1704.42  3760.9 1705.26
  4608.6 1709.95  4648.8 1708.28  4668.9 1701.53  4699.0 1697.73  4725.9 1702.83
  4910.0 1701.11  4943.3 1704.86  4970.2 1698.57  4978.1 1691.48  4981.1 1690.18
  5014.1 1691.48  5020.4 1702.31  5060.6 1703.09  5120.9 1709.77  5361.1 1707.35
  6540.2 1707.95  6679.6 1705.23  7433.3 1717.80  7953.6 1739.76  8223.8 1737.25
  8333.9 1741.41  8404.0 1738.48  8644.1 1743.13  8754.2 1747.74  8784.5 1759.68
#Mann=3,-1,0
  -356.1    0.05       0  4978.1    0.05       0  5014.1    0.05       0
Bank Sta=4978.1,5014.1
Exp/Cntr=0.3,0.1

Type RM Length L Ch R = 1,634677,488,488,488
BEGIN DESCRIPTION:
Mapping XS cf996e9b
END DESCRIPTION:
XS GIS Cut Line= 4
      1513470.49      6931485.81      1513244.82      6931173.34
      1513244.82      6930426.81      1514842.04      6923308.78
#Sta/Elev= 30
    60.7 1716.38   400.2 1716.44   446.1 1714.28   651.5 1716.47  1260.0 1708.72
  2062.6 1702.68  2103.6 1704.60  2448.2 1705.11  2902.0 1703.28  4867.9 1706.35
  4911.2 1704.55  4932.2 1699.48  4959.7 1698.50  4977.5 1690.17  4981.3 1688.87
  5022.5 1690.17  5024.4 1693.33  5034.7 1697.78  5044.9 1699.00  5185.2 1698.24
  5270.4 1694.55  5283.5 1698.04  5297.0 1698.40  5326.8 1700.18  5332.0 1702.86
  5393.4 1706.01  6379.9 1705.82  6828.2 1708.30  8191.3 1726.17  8487.7 1725.59
#Mann=5,-1,0
    60.7    0.05       0  4977.5   0.035       0  5022.5    0.05       0
  5185.2     0.1       0  5297.0    0.05       0
Bank Sta=4977.5,5022.5
Exp/Cntr=0.3,0.1

Type RM Length L Ch R = 1,634189,2015,2015,2015
BEGIN DESCRIPTION:
Mapping XS c2ac677d
END DESCRIPTION:
XS GIS Cut Line= 3
      1513574.68      6930982.32      1513592.04      6930357.37
      1515310.41      6923067.34
#Sta/Elev= 30
  1023.1 1715.21  1567.6 1713.87  2315.5 1706.55  2664.8 1700.50  2725.2 1702.83
  3206.3 1703.63  3476.4 1700.79  3513.0 1702.80  4853.1 1705.89  4903.9 1700.54
  4909.0 1697.85  4951.4 1697.64  4956.5 1690.50  4966.0 1687.19  4969.0 1685.89
  5002.0 1687.19  5007.3 1695.77  5017.5 1697.74  5202.5 1696.25  5284.7 1704.81
  6479.6 1703.69  7087.7 1707.74  8266.8 1720.88  8366.8 1722.02  8455.7 1722.96
  8566.6 1723.93  8642.9 1725.58  8766.5 1729.91  8922.6 1734.66  9138.1 1735.37
#Mann=9,-1,0
  1023.1    0.05       0  4966.0    0.05       0  5002.0    0.05       0
  8266.8    0.12       0  8366.8    0.05       0  8455.7    0.12       0
  8566.6    0.05       0  8642.9    0.12       0  8766.5    0.05       0
Bank Sta=4966,5002
Exp/Cntr=0.3,0.1

Type RM Length L Ch R = 1,632174,2991,2991,2991
BEGIN DESCRIPTION:
Mapping XS f3615e49
END DESCRIPTION:
XS GIS Cut Line= 4
      1515090.39      6932021.06      1516027.90      6928843.94
      1515194.57      6925692.90      1515663.32      6923166.85
#Sta/Elev= 30
   559.0 1713.56  2866.4 1712.85  4260.4 1702.02  4945.7 1704.63  4974.1 1697.05
  4990.3 1686.93  4994.0 1685.63  5035.3 1686.93  5039.1 1691.51  5056.9 1695.64
  5119.5 1691.40  5207.1 1696.29  5275.3 1704.11  7130.9 1702.36  8549.6 1713.17
  8754.2 1716.37  8917.7 1726.82  9037.8 1728.25  9119.2 1736.26  9210.7 1755.39
  9231.1 1755.17  9261.6 1746.28  9297.7 1749.73  9363.3 1738.65  9403.4 1738.12
  9514.1 1750.50  9519.2 1748.06  9572.0 1759.10  9658.3 1754.88  9700.1 1759.66
#Mann=5,-1,0
   559.0    0.05       0  4945.7     0.1       0  4990.3    0.07       0
  5035.3     0.1       0  5207.1    0.05       0
Bank Sta=4990.3,5035.3
Exp/Cntr=0.3,0.1

Type RM Length L Ch R = 1,629183,2222,2222,2222
BEGIN DESCRIPTION:
Mapping XS f19cea20
END DESCRIPTION:
XS GIS Cut Line= 3
      1519705.40      6932412.82      1519346.04      6929033.64
      1516289.17      6923116.43
#Sta/Elev= 30
 -1044.1 1713.47  -576.7 1708.28  2632.5 1709.39  4309.9 1699.32  4802.4 1701.75
  4808.0 1694.13  4824.6 1687.04  4896.6 1688.63  4955.7 1682.60  4960.9 1681.30
  5018.7 1682.60  5023.9 1689.23  5046.0 1694.97  5388.2 1692.12  5534.6 1701.06
  6551.8 1700.19  7144.2 1693.04  7963.3 1705.06  8255.3 1713.14  8340.0 1716.00
  8467.2 1736.10  8533.7 1727.37  8607.3 1731.99  8705.2 1748.76  8733.0 1759.49
  8771.7 1756.58  8799.5 1764.58  8854.7 1755.06  8926.7 1766.72  9014.3 1764.48
#Mann=5,-1,0
 -1044.1    0.05       0  4955.7    0.05       0  5018.7    0.05       0
  7963.3    0.12       0  8255.3    0.05       0
Bank Sta=4955.7,5018.7
Exp/Cntr=0.3,0.1

Type RM Length L Ch R = 1,626961,8251,8251,8251
BEGIN DESCRIPTION:
Mapping XS 2b30422f
END DESCRIPTION:
XS GIS Cut Line= 5
      1522179.35      6931414.51      1521507.61      6927884.52
      1520168.53      6925771.02      1518632.07      6924494.98
      1517173.76      6922125.22
#Sta/Elev= 30
 -1575.1 1705.11  3674.2 1709.00  3851.3 1709.44  3870.8 1709.44  4066.2 1709.69
  4423.6 1700.12  4943.5 1700.02  4972.2 1693.12  4977.9 1679.90  4981.7 1678.60
  5022.9 1679.90  5029.5 1688.84  5051.4 1691.38  5082.1 1689.35  5257.6 1691.21
  5398.9 1692.11  5461.8 1701.13  6384.9 1697.06  6491.7 1687.52  6541.9 1696.95
  7167.9 1690.83  7919.5 1698.83  8148.1 1704.68  8592.2 1710.03  8789.0 1727.89
  8874.1 1745.13  8999.6 1742.61  9160.9 1756.97  9296.9 1761.95  9300.0 1761.95
#Mann=15,-1,0
 -1575.1    0.05       0  3674.2     0.1       0  3851.3    0.05       0
  3870.8     0.1       0  4066.2    0.05       0  4977.9    0.05       0
  5022.9    0.05       0  5051.4    0.12       0  5082.1    0.05       0
  5257.6    0.12       0  5398.9    0.05       0  7919.5    0.12       0
  8148.1    0.05       0  9160.9    0.12       0  9296.9    0.05       0
Bank Sta=4977.9,5022.9
Exp/Cntr=0.3,0.1

Type RM Length L Ch R = 1,618710,3037,3037,3037
BEGIN DESCRIPTION:
Mapping XS d7c8b0c1
END DESCRIPTION:
XS GIS Cut Line= 5
      1523196.29      6928754.03      1523231.01      6927695.03
      1521546.98      6923580.44      1519307.40      6922781.83
      1518751.82      6921306.09
#Sta/Elev= 30
 -3616.7 1701.94 -1817.7 1706.73  -658.8 1693.09   582.9 1699.78   743.1 1694.97
  4258.0 1695.89  4603.4 1693.93  4658.5 1687.29  4939.3 1685.48  4964.2 1684.24
  4977.5 1678.14  4981.3 1677.14  5022.5 1678.14  5024.6 1684.99  5039.9 1695.70
  5071.9 1704.15  5134.8 1691.67  5178.8 1700.26  5195.2 1699.12  5200.6 1703.56
  5274.9 1696.05  5310.8 1708.13  5365.9 1702.13  5371.2 1706.95  5381.8 1705.20
  5413.9 1713.60  5676.9 1724.52  5707.1 1710.47  5737.4 1706.49  5843.3 1709.42
#Mann=3,-1,0
 -3616.7    0.05       0  4977.5    0.05       0  5022.5    0.05       0
Bank Sta=4977.5,5022.5
Exp/Cntr=0.3,0.1

Type RM Length L Ch R = 1,615673,2689,2689,2689
BEGIN DESCRIPTION:
Mapping XS f2fc6cd0
END DESCRIPTION:
XS GIS Cut Line= 3
      1523533.43      6932367.83      1523411.90      6927506.76
      1520095.91      6919815.74
#Sta/Elev= 30
 -4895.4 1710.79 -2034.7 1701.53   626.7 1706.52  1479.5 1695.11  2977.3 1697.76
  4829.3 1693.40  4976.8 1682.48  4986.7 1672.77  4990.5 1671.47  5031.7 1672.77
  5062.3 1677.81  5070.9 1684.55  5076.3 1680.04  5099.9 1685.63  5146.9 1680.91
  5293.0 1691.24  5400.9 1692.27  5476.8 1692.54  5508.7 1692.65  6462.4 1696.69
  7131.4 1707.04  7164.0 1712.18  7217.0 1708.81  7360.1 1712.63  7474.0 1726.75
  7534.3 1724.55  7643.2 1746.05  8000.5 1750.91  8097.5 1747.72  8342.6 1757.58
#Mann=9,-1,0
 -4895.4    0.05       0  4829.3     0.1       0  4986.7    0.07       0
  5031.7     0.1       0  5293.0     0.1       0  5400.9    0.05       0
  5476.8     0.1       0  5508.7    0.05       0  8097.5    0.12       0
Bank Sta=4986.7,5031.7
Exp/Cntr=0.3,0.1

Type RM Length L Ch R = 1,612984,3915,3915,3915
BEGIN DESCRIPTION:
Mapping XS 58148f4d
END DESCRIPTION:
XS GIS Cut Line= 2
      1525611.24      6929703.34      1522902.89      6920093.91
#Sta/Elev= 30
 -1499.3 1709.72  -922.3 1700.23   315.4 1696.13   535.1 1699.59  3711.4 1703.13
  4230.9 1700.17  4773.1 1690.36  4854.3 1684.96  4887.5 1688.24  4920.6 1690.18
  4959.8 1682.61  4986.4 1671.08  4988.7 1669.78  5013.4 1671.08  5020.5 1681.17
  5051.7 1684.47  5174.3 1680.05  5233.8 1682.39  5292.0 1689.12  5997.1 1685.42
  7127.8 1689.15  7459.9 1684.18  7823.5 1693.35  8075.1 1711.41  8116.3 1723.89
  8158.2 1737.25  8236.6 1743.68  8383.1 1746.36  8449.1 1743.52  8484.5 1733.61
#Mann=8,-1,0
 -1499.3    0.05       0  4773.1    0.12       0  4887.5     0.1       0
  4986.4    0.07       0  5013.4     0.1       0  5233.8    0.05       0
  7823.5    0.12       0  8116.3    0.05       0
Bank Sta=4986.4,5013.4
Exp/Cntr=0.3,0.1

Type RM Length L Ch R = 1,609069,2141,2141,2141
BEGIN DESCRIPTION:
Clear Fork Brazos Rv 144.0
END DESCRIPTION:
XS GIS Cut Line= 4
      1525366.65      6926890.96      1526114.61      6924298.52
      1525255.00      6920538.00      1525255.00      6920038.00
#Sta/Elev= 30
 -1561.0 1698.36  1140.0 1698.29  2462.7 1694.00  2532.8 1689.91  3240.6 1683.86
  4327.9 1689.20  4369.0 1685.42  4658.1 1685.38  4759.1 1685.35  4810.1 1685.02
  4879.6 1676.88  4962.4 1678.59  4994.7 1678.43  4994.9 1667.76  4998.6 1666.46
  5039.9 1667.76  5054.7 1678.69  5074.7 1681.97  5108.5 1699.72  5134.7 1710.03
  5174.7 1706.12  5204.7 1715.34  5264.7 1710.41  5294.7 1716.33  5314.7 1708.00
  5334.7 1706.22  5364.7 1717.92  5404.7 1717.62  5424.7 1727.64  5494.7 1733.72
#Mann=7,-1,0
 -1561.0    0.05       0  4658.1     0.1       0  4759.1    0.05       0
  4962.4     0.1       0  4994.9    0.07       0  5039.9     0.1       0
  5108.5    0.05       0
Bank Sta=4994.9,5039.9
Exp/Cntr=0.3,0.1

Type RM Length L Ch R = 1,606928,2419,2419,2419
BEGIN DESCRIPTION:
Mapping XS 0342b55d
END DESCRIPTION:
XS GIS Cut Line= 3
      1525874.46      6925875.35      1527799.72      6922338.22
      1526658.44      6919086.64
#Sta/Elev= 30
  -904.8 1697.69  1179.5 1695.59  3331.1 1681.31  4756.0 1686.49  4900.4 1685.22
  4962.4 1673.43  4987.8 1676.87  4992.6 1665.33  4996.4 1664.03  5037.6 1665.33
  5055.3 1676.21  5205.0 1677.42  5261.7 1686.72  5385.7 1685.88  5418.3 1691.47
  5509.7 1714.58  5602.6 1716.38  5623.0 1722.69  5644.9 1723.63  5666.1 1723.03
  5690.3 1716.02  5783.3 1718.55  5809.0 1724.83  5888.7 1723.54  5920.5 1727.83
  6175.6 1723.93  6196.0 1730.48  6227.0 1732.39  6351.0 1726.65  6568.4 1726.66
#Mann=5,-1,0
  -904.8    0.05       0  4756.0     0.1       0  4992.6    0.07       0
  5037.6     0.1       0  5418.3    0.05       0
Bank Sta=4992.6,5037.6
Exp/Cntr=0.3,0.1

Type RM Length L Ch R = 1,604509,336,336,336
BEGIN DESCRIPTION:
Mapping XS a9f59c11
END DESCRIPTION:
XS GIS Cut Line= 6
      1528479.45      6926099.93      1528798.21      6923199.15
      1529172.75      6922003.51      1529201.56      6919208.86
      1529885.66      6917084.76      1529359.83      6916203.23
#Sta/Elev= 30
  -826.9 1707.76  -161.0 1694.84   180.6 1691.01   463.8 1690.46   513.1 1688.65
   828.0 1688.43  1126.7 1683.98  1288.2 1686.59  3134.8 1683.50  3390.0 1680.57
  3460.2 1683.61  4558.3 1681.36  4895.7 1683.96  4915.8 1682.53  4945.9 1674.82
  4974.8 1672.66  4977.5 1663.21  4981.3 1662.21  5022.5 1663.21  5026.1 1674.13
  5066.2 1672.49  5096.3 1673.93  5126.4 1680.59  5597.9 1684.23  6915.0 1680.66
  7180.8 1683.51  8781.6 1686.46  9379.5 1693.95  9392.7 1696.55  9408.3 1694.99
#Mann=3,-1,0
  -826.9    0.05       0  4977.5    0.05       0  5022.5    0.05       0
Bank Sta=4977.5,5022.5
Exp/Cntr=0.3,0.1

Type RM Length L Ch R = 1,604173,3565,3565,3565
BEGIN DESCRIPTION:
Mapping XS bebd9566
END DESCRIPTION:
XS GIS Cut Line= 6
      1528726.01      6926109.78      1528798.21      6924826.96
      1529576.10      6921873.86      1529504.08      6919698.65
      1530138.42      6917265.30      1529349.59      6915996.99
#Sta/Elev= 30
  -982.3 1708.51  -700.1 1706.88  -201.9 1693.97   806.3 1689.00  1285.4 1683.42
  3063.2 1684.26  3310.9 1679.32  3583.5 1683.72  4276.8 1679.69  4751.6 1683.93
  4833.5 1681.07  4854.7 1676.41  4890.0 1673.17  4941.3 1673.95  4971.7 1673.93
  4977.5 1663.65  4981.3 1662.65  5022.5 1663.65  5030.7 1674.07  5048.8 1678.07
  5099.8 1682.49  5345.0 1683.90  6162.2 1680.21  6482.6 1683.09  6697.9 1676.93
  6715.2 1680.04  6923.8 1685.49  8798.3 1685.88  9370.9 1693.51  9557.8 1698.75
#Mann=7,-1,0
  -982.3    0.05       0  4751.6     0.1       0  4854.7    0.05       0
  4941.3     0.1       0  4977.5    0.07       0  5022.5     0.1       0
  5048.8    0.05       0
Bank Sta=4977.5,5022.5
Exp/Cntr=0.3,0.1

Type RM Length L Ch R = 1,600608,4631,4631,4631
BEGIN DESCRIPTION:
Mapping XS 5f017d27
END DESCRIPTION:
XS GIS Cut Line= 3
      1533195.86      6922298.78      1531481.46      6919347.41
      1529159.69      6915419.93
#Sta/Elev= 30
   476.2 1701.31   886.8 1701.45  1517.6 1670.49  1625.2 1676.00  2534.2 1680.59
  3125.4 1678.81  4434.7 1682.24  4466.8 1678.70  4537.5 1679.06  4564.3 1674.71
  4697.0 1668.33  4718.4 1672.56  4739.9 1667.81  4776.9 1671.81  4927.3 1671.04
  4945.8 1670.58  4958.3 1661.47  4965.5 1660.15  4968.5 1658.85  5001.5 1660.15
  5003.9 1671.80  5018.6 1676.47  5053.9 1680.51  5223.6 1678.68  7230.7 1685.78
  7529.1 1690.64  7566.1 1694.53  7667.5 1692.28  7997.2 1702.16  8451.8 1703.86
#Mann=7,-1,0
   476.2    0.05       0  4466.8     0.1       0  4537.5    0.05       0
  4927.3     0.1       0  4965.5    0.07       0  5001.5     0.1       0
  5018.6    0.05       0
Bank Sta=4965.5,5001.5
Exp/Cntr=0.3,0.1

Type RM Length L Ch R = 1,595977,2889,2889,2889
BEGIN DESCRIPTION:
Mapping XS ac20b5de
END DESCRIPTION:
XS GIS Cut Line= 3
      1534531.54      6921340.81      1533537.58      6917681.90
      1532831.72      6915434.67
#Sta/Elev= 30
  2355.0 1699.45  2492.6 1697.58  2679.2 1687.35  2784.2 1686.87  2927.8 1677.95
  3166.6 1670.41  3228.4 1663.82  3235.9 1667.56  3259.4 1671.30  3355.3 1675.24
  4015.9 1678.05  4194.6 1675.41  4409.7 1678.63  4502.9 1675.62  4731.0 1675.74
  4845.2 1667.25  4954.2 1667.22  4969.2 1665.80  4982.0 1657.22  4985.0 1656.22
  5018.0 1657.22  5021.1 1667.58  5041.8 1672.89  5068.4 1677.69  5103.1 1678.11
  5679.3 1673.22  7669.3 1671.85  7874.3 1672.57  8106.4 1679.81  8502.0 1679.08
#Mann=3,-1,0
  2355.0    0.05       0  4982.0    0.05       0  5018.0    0.05       0
Bank Sta=4982,5018
Exp/Cntr=0.3,0.1

Type RM Length L Ch R = 1,593088,4066,4066,4066
BEGIN DESCRIPTION:
Mapping XS 0403abc8
END DESCRIPTION:
XS GIS Cut Line= 3
      1536451.07      6921343.89      1535995.35      6918110.43
      1532392.90      6914095.65
#Sta/Elev= 30
  3528.5 1702.30  4332.3 1699.99  4468.1 1691.98  4610.5 1679.40  4645.3 1682.26
  4675.6 1681.02  4705.9 1686.47  4752.8 1687.92  4867.5 1679.25  4900.3 1673.87
  4943.6 1665.45  4971.4 1663.73  4978.6 1661.06  4981.5 1654.54  4984.5 1653.24
  5017.5 1654.54  5019.0 1660.18  5029.1 1665.43  5089.7 1666.49  5140.2 1674.84
  6792.6 1670.28  7879.4 1670.61  8693.4 1667.55  8884.8 1664.45  9522.5 1676.54
  9982.2 1680.43 10393.4 1677.53 11696.3 1683.43 11710.5 1681.41 12188.0 1682.32
#Mann=5,-1,0
  3528.5    0.05       0  4900.3     0.1       0  4943.6    0.05       0
  4981.5   0.035       0  5017.5    0.05       0
Bank Sta=4981.5,5017.5
Exp/Cntr=0.3,0.1

Type RM Length L Ch R = 1,589022,4637,4637,4637
BEGIN DESCRIPTION:
Mapping XS 74d5c278
END DESCRIPTION:
XS GIS Cut Line= 4
      1540357.30      6920410.76      1538794.83      6919521.02
      1536581.29      6918631.26      1532676.10      6913901.65
#Sta/Elev= 30
  4249.1 1694.81  4896.6 1692.58  4949.9 1673.80  4977.3 1667.07  4987.4 1659.82
  4989.2 1651.97  4991.5 1650.67  5016.2 1651.97  5022.8 1653.05  5030.6 1659.04
  5036.4 1660.58  5073.8 1662.49  5095.4 1660.14  5170.4 1670.88  5851.3 1669.03
  6065.9 1671.96  7815.7 1669.43  8318.3 1671.68  8401.6 1669.71 10087.2 1670.74
 10393.4 1667.78 10719.5 1668.12 10819.4 1662.74 11017.7 1669.20 11856.5 1680.37
 12673.3 1676.39 13965.7 1680.45 14037.4 1682.31 14058.2 1680.26 14566.3 1681.79
#Mann=3,-1,0
  4249.1    0.05       0  4989.2    0.05       0  5016.2    0.05       0
Bank Sta=4989.2,5016.2
Exp/Cntr=0.3,0.1

Type RM Length L Ch R = 1,584385,2224,2224,2224
BEGIN DESCRIPTION:
Mapping XS c52d7704
END DESCRIPTION:
XS GIS Cut Line= 4
      1540769.03      6918978.36      1539098.05      6918085.25
      1536548.30      6917782.73      1534329.96      6915405.94
#Sta/Elev= 30
   880.8 1693.60  1039.6 1691.58  1335.5 1672.77  1533.0 1667.48  3141.1 1670.19
  4178.3 1665.11  4581.6 1667.89  4611.3 1664.48  4702.0 1663.28  4792.6 1656.86
  4829.7 1658.24  4873.1 1656.03  4903.4 1660.48  4963.8 1660.59  4973.8 1658.17
  4982.0 1648.98  4985.0 1647.98  5018.0 1648.98  5044.3 1661.49  5064.5 1666.06
  5170.7 1669.64  6544.5 1668.75  6629.5 1666.99  6657.8 1662.02  6686.1 1661.57
  7174.2 1675.37  7415.0 1674.71  7527.9 1678.53  7959.7 1674.94  8594.3 1674.44
#Mann=3,-1,0
   880.8    0.05       0  4982.0    0.05       0  5018.0    0.05       0
Bank Sta=4982,5018
Exp/Cntr=0.3,0.1

Type RM Length L Ch R = 1,582161,5786,5786,5786
BEGIN DESCRIPTION:
Clear Fork Brazos Rv 141.0
END DESCRIPTION:
XS GIS Cut Line= 3
      1540805.01      6918738.01      1538305.00      6917238.00
      1535135.07      6912773.02
#Sta/Elev= 30
  2084.4 1691.75  2368.2 1674.00  2601.4 1666.80  4519.8 1668.63  4780.3 1666.58
  4832.7 1658.98  4864.6 1657.98  4949.4 1658.00  4979.4 1646.79  4981.6 1645.49
  5006.4 1646.79  5007.3 1654.75  5028.2 1657.27  5085.7 1655.88  5099.5 1657.85
  5161.6 1657.83  5236.1 1661.21  5271.7 1666.09  5320.2 1665.47  5406.5 1667.11
  6706.1 1665.11  7244.2 1661.08  7581.9 1663.54  7739.4 1668.05  8027.2 1668.04
  8398.7 1674.39  8965.8 1674.61  9467.7 1679.39 10055.7 1681.44 10475.7 1680.74
#Mann=7,-1,0
  2084.4    0.05       0  4864.6     0.1       0  4979.4    0.07       0
  5006.4     0.1       0  5161.6    0.05       0  5320.2     0.1       0
  5406.5    0.05       0
Bank Sta=4979.4,5006.4
Exp/Cntr=0.3,0.1

Type RM Length L Ch R = 1,576375,4782,4782,4782
BEGIN DESCRIPTION:
Mapping XS bee2ba9b
END DESCRIPTION:
XS GIS Cut Line= 3
      1542724.12      6917683.38      1541203.25      6915995.85
      1537765.73      6911495.82
#Sta/Elev= 30
  3820.9 1689.20  4312.8 1686.72  4525.3 1676.35  4574.6 1677.05  4645.6 1671.86
  4881.7 1665.14  4925.5 1663.78  4949.8 1662.91  4964.0 1658.15  4978.2 1652.52
  4979.0 1642.62  4982.0 1641.32  5015.0 1642.62  5020.8 1653.20  5041.1 1654.08
  5473.7 1655.14  5530.5 1652.98  5565.6 1648.25  5742.7 1656.78  5785.3 1662.05
  6117.9 1664.86  6240.5 1662.59  6668.5 1664.83  8915.0 1663.09  9093.7 1657.42
  9199.7 1658.50  9264.1 1662.81 10342.5 1664.52 10941.1 1674.30 11755.4 1674.90
#Mann=6,-1,0
  3820.9    0.05       0  4881.7     0.1       0  4925.5    0.05       0
  4979.0    0.07       0  5015.0    0.05       0  5041.1    0.05       0
Bank Sta=4979,5015
Exp/Cntr=0.3,0.1

Type RM Length L Ch R = 1,571593,1735,1735,1735
BEGIN DESCRIPTION:
Clear Fork Brazos Rv 139.0
END DESCRIPTION:
XS GIS Cut Line= 3
      1543805.03      6915638.04      1542122.93      6913250.46
      1539304.98      6912137.99
#Sta/Elev= 30
  2063.2 1682.18  2522.7 1678.15  2823.2 1667.93  3017.4 1658.47  3147.1 1655.65
  3203.8 1657.55  3605.3 1660.25  4202.7 1662.03  4467.5 1658.94  4833.3 1661.07
  4848.1 1660.73  4889.9 1650.92  4925.7 1646.98  4955.2 1649.71  4976.1 1648.66
  4982.3 1646.54  4988.4 1639.96  4990.6 1638.66  5015.4 1639.96  5024.6 1646.71
  5030.7 1648.50  5175.1 1653.52  5207.4 1659.53  5222.7 1659.91  5301.2 1658.80
  5562.1 1662.03  5701.9 1660.24  5985.7 1661.81  7457.4 1661.67  8013.4 1669.99
#Mann=3,-1,0
  2063.2    0.05       0  4988.4   0.035       0  5015.4    0.05       0
Bank Sta=4988.4,5015.4
Exp/Cntr=0.3,0.1

Type RM Length L Ch R = 1,569858,3093,3093,3093
BEGIN DESCRIPTION:
Mapping XS 43527efd
END DESCRIPTION:
XS GIS Cut Line= 4
      1545133.92      6915204.20      1543491.69      6912409.53
      1540380.13      6911041.02      1538400.47      6910588.91
#Sta/Elev= 30
  1752.7 1671.73  2114.7 1659.43  2450.6 1655.92  3970.3 1657.96  4759.4 1661.81
  4796.5 1660.02  4823.8 1650.32  4839.5 1648.05  4949.5 1647.85  4956.7 1638.87
  4962.5 1637.92  4966.3 1636.92  5007.5 1637.92  5008.7 1647.45  5014.1 1648.01
  5274.6 1652.49  5357.3 1656.37  5404.0 1661.04  6572.2 1659.55  6793.1 1656.56
  6967.5 1660.59  7292.8 1661.68  9680.8 1662.02 10136.7 1669.87 10162.9 1674.16
 10214.2 1668.34 10270.7 1671.94 10337.3 1670.34 10368.1 1673.65 10424.0 1674.23
#Mann=3,-1,0
  1752.7    0.05       0  4962.5    0.05       0  5007.5    0.05       0
Bank Sta=4962.5,5007.5
Exp/Cntr=0.3,0.1

Type RM Length L Ch R = 1,566765,3831,3831,3831
BEGIN DESCRIPTION:
Clear Fork Brazos Rv 138.0
END DESCRIPTION:
XS GIS Cut Line= 3
      1546767.02      6914747.84      1545855.00      6912338.00
      1544355.00      6907338.00
#Sta/Elev= 30
  2420.4 1667.34  3532.2 1666.10  3935.4 1650.30  4726.5 1659.77  4751.1 1658.70
  4793.9 1645.52  4826.0 1643.25  4899.7 1645.04  4975.7 1644.36  4982.0 1641.04
  4987.3 1641.79  4989.5 1636.10  4992.5 1634.70  5025.5 1636.10  5046.6 1644.60
  5079.7 1652.76  5084.9 1650.39  5117.0 1658.60  6281.2 1655.74  6854.6 1658.31
  7002.5 1652.36  7167.8 1657.86  7794.2 1654.91  8745.1 1655.76  8810.4 1653.40
  9632.5 1657.00  9854.4 1660.62  9966.6 1665.81 10008.4 1672.74 10217.2 1679.61
#Mann=5,-1,0
  2420.4    0.05       0  4899.7     0.1       0  4989.5    0.07       0
  5025.5     0.1       0  5117.0    0.05       0
#XS Ineff=2,0
       0                 6278.50    0.00 1671.44
Permanent Ineff=
       F       F
Bank Sta=4989.5,5025.5
Exp/Cntr=0.3,0.1

Type RM Length L Ch R = 1,562934,4438,4438,4438
BEGIN DESCRIPTION:
Clear Fork Brazos Rv 137.0
END DESCRIPTION:
XS GIS Cut Line= 3
      1547605.00      6913938.02      1547605.00      6911438.00
      1545605.02      6906938.04
#Sta/Elev= 30
  2498.1 1665.43  3098.1 1658.98  3478.1 1651.19  3818.1 1648.77  4018.1 1653.52
  4918.1 1656.08  4928.1 1655.62  4977.2 1633.26  4980.2 1631.86  5013.2 1633.26
  5030.3 1643.48  5173.2 1642.67  5238.9 1654.92  5271.7 1656.72  6831.8 1655.24
  7132.7 1650.64  7376.2 1654.77  8992.4 1650.58  9444.5 1654.22  9594.9 1657.67
  9747.5 1671.35  9786.4 1682.01  9832.9 1691.05  9838.4 1689.70  9856.2 1695.63
  9861.7 1693.87  9884.9 1704.67  9890.4 1703.12  9908.2 1710.27  9922.5 1712.24
#Mann=3,-1,0
  2498.1    0.05       0  4977.2    0.04       0  5013.2    0.05       0
#XS Ineff=2,0
       0                 6607.10    0.00 1681.07
Permanent Ineff=
       F       F
Bank Sta=4977.2,5013.2
Exp/Cntr=0.3,0.1

Type RM Length L Ch R = 1,558496,3312,3312,3312
BEGIN DESCRIPTION:
Mapping XS ada4a363
END DESCRIPTION:
XS GIS Cut Line= 3
      1550252.17      6915770.62      1549453.25      6908975.01
      1548329.11      6906705.91
#Sta/Elev= 30
 -2625.0 1678.90 -1838.8 1658.32 -1625.5 1663.87 -1565.1 1658.12  -552.1 1651.15
  1324.6 1647.58  4715.5 1652.15  4805.2 1640.99  4961.8 1640.81  4975.4 1630.64
  4979.1 1629.24  5020.4 1630.64  5028.7 1646.60  5040.6 1651.28  5185.0 1659.66
  5421.8 1654.83  5578.7 1657.42  5609.1 1666.66  5662.8 1657.09  5803.0 1663.73
  5937.5 1689.35  5976.8 1704.21  6066.5 1699.92  6279.4 1706.69  6341.1 1693.53
  6414.0 1687.98  6453.2 1698.58  6468.4 1695.18  6513.0 1708.12  6749.7 1708.77
#Mann=3,-1,0
 -2625.0    0.05       0  4975.4    0.05       0  5020.4    0.05       0
Bank Sta=4975.4,5020.4
Exp/Cntr=0.3,0.1

Type RM Length L Ch R = 1,555184,3537,3537,3537
BEGIN DESCRIPTION:
Clear Fork Brazos Rv 135.0
END DESCRIPTION:
XS GIS Cut Line= 3
      1552539.59      6916093.32      1551955.00      6908638.00
      1551955.00      6907638.00
#Sta/Elev= 30
 -2477.6 1678.98 -2231.7 1668.71 -1850.4 1661.83 -1248.5 1656.22  2322.4 1651.37
  2773.8 1645.99  2864.1 1641.43  3074.7 1647.12  3706.6 1645.74  4659.6 1648.28
  4830.1 1646.88  4890.3 1640.45  4960.5 1637.70  4968.2 1634.30  4980.7 1631.78
  4982.9 1630.38  5007.7 1631.78  5010.6 1634.39  5040.6 1638.30  5090.6 1650.11
  5164.1 1648.76  5530.6 1649.27  5580.6 1651.63  5653.6 1663.57  5710.6 1683.50
  5751.5 1693.35  5800.6 1698.73  5870.6 1695.76  5920.6 1698.28  6000.6 1697.34
#Mann=7,-1,0
 -2477.6    0.05       0  4968.2     0.1       0  4980.7    0.07       0
  5007.7     0.1       0  5164.1    0.05       0  5653.6    0.12       0
  5751.5    0.05       0
Bank Sta=4980.7,5007.7
Exp/Cntr=0.3,0.1

Type RM Length L Ch R = 1,551647,2564,2564,2564
BEGIN DESCRIPTION:
Mapping XS 12294fab
END DESCRIPTION:
XS GIS Cut Line= 2
      1555786.59      6915391.71      1553974.08      6907287.52
#Sta/Elev= 30
 -2696.0 1670.84 -2617.7 1671.41 -2341.9 1663.44 -1595.8 1658.51  -796.5 1658.13
   -28.0 1652.61  1703.8 1651.50  2006.8 1643.93  2239.2 1643.80  2349.4 1640.32
  4685.7 1647.32  4716.4 1641.41  4788.1 1635.25  4947.6 1636.57  4972.6 1636.33
  4976.7 1629.41  4979.7 1628.01  5012.7 1629.41  5013.6 1633.57  5034.5 1634.70
  5078.7 1637.51  5105.8 1646.23  5198.0 1661.76  5236.4 1673.72  5290.3 1696.53
  5385.8 1696.07  5433.7 1690.06  5484.7 1671.34  5538.4 1691.69  5608.4 1695.07
#Mann=7,-1,0
 -2696.0    0.05       0  4947.6     0.1       0  4976.7    0.07       0
  5012.7     0.1       0  5034.5    0.05       0  5236.4    0.12       0
  5385.8    0.05       0
Bank Sta=4976.7,5012.7
Exp/Cntr=0.3,0.1

Type RM Length L Ch R = 1,549083,2639,2639,2639
BEGIN DESCRIPTION:
Mapping XS 536539a4
END DESCRIPTION:
XS GIS Cut Line= 4
      1556269.31      6912643.94      1556283.65      6911372.35
      1556326.87      6907540.52      1556168.41      6906186.41
#Sta/Elev= 30
    16.3 1651.68  1242.3 1650.82  1582.3 1648.36  1810.8 1641.82  1882.4 1638.99
  2004.1 1641.12  4802.5 1645.80  4862.6 1635.21  4942.6 1634.18  4962.6 1625.01
  4972.0 1624.72  4975.0 1623.72  5008.0 1624.72  5012.6 1633.52  5022.6 1630.80
  5052.6 1633.37  5142.7 1631.82  5162.9 1634.67  5439.1 1637.60  5539.7 1640.56
  5746.8 1646.21  5998.5 1648.96  6028.7 1650.54  6048.9 1654.76  6208.3 1648.56
  6320.7 1649.36  6350.9 1653.06  6461.7 1649.84  6473.2 1653.57  6483.4 1653.43
#Mann=7,-1,0
    16.3    0.05       0  1810.8    0.12       0  2004.1    0.05       0
  4972.0    0.05       0  5008.0    0.05       0  5439.1     0.1       0
  5539.7    0.05       0
Bank Sta=4972,5008
Exp/Cntr=0.3,0.1

Type RM Length L Ch R = 1,546444,1164,1164,1164
BEGIN DESCRIPTION:
Mapping XS a53f048e
END DESCRIPTION:
XS GIS Cut Line= 3
      1557974.08      6914308.35      1558570.44      6908282.31
      1558133.14      6905741.84
#Sta/Elev= 30
 -1911.5 1670.33 -1378.6 1668.31  -227.4 1657.09    18.2 1657.42   329.7 1643.81
   570.9 1641.17  4040.4 1639.00  4899.2 1644.30  4913.7 1643.50  4950.0 1631.26
  4973.6 1631.02  4978.2 1621.21  4981.2 1619.81  5014.2 1621.21  5021.0 1631.23
  5041.3 1632.19  5088.3 1644.32  5761.7 1642.58  6157.5 1637.55  6370.6 1641.23
  6446.1 1649.14  6501.0 1661.41  6506.0 1659.51  6560.9 1673.00  6566.0 1670.58
  6603.9 1682.71  6620.8 1683.83  6625.9 1680.38  6675.0 1684.35  6721.8 1683.16
#Mann=3,-1,0
 -1911.5    0.05       0  4978.2    0.05       0  5014.2    0.05       0
Bank Sta=4978.2,5014.2
Exp/Cntr=0.3,0.1

Type RM Length L Ch R = 1,545280,3834,3834,3834
BEGIN DESCRIPTION:
Mapping XS 12989441
END DESCRIPTION:
XS GIS Cut Line= 4
      1562023.02      6910874.82      1560338.98      6909850.51
      1559470.93      6907038.01      1558203.59      6905544.97
#Sta/Elev= 30
   348.2 1648.44  1799.0 1650.10  1879.2 1652.90  1909.4 1650.24  1946.2 1653.27
  1983.0 1649.89  2484.8 1649.47  2949.8 1639.08  3370.3 1636.37  4844.1 1642.67
  4954.1 1630.99  4962.6 1630.62  4977.3 1621.31  4978.0 1621.07  4981.0 1619.67
  5014.0 1621.07  5022.0 1631.23  5053.4 1630.71  5137.1 1642.98  6451.9 1640.43
  6501.3 1634.82  6792.4 1642.81  6934.1 1660.51  6948.4 1659.50  7012.1 1674.91
  7019.8 1672.30  7026.3 1675.37  7040.6 1668.64  7112.1 1659.75  7221.1 1664.14
#Mann=5,-1,0
   348.2    0.05       0  4954.1     0.1       0  4977.3    0.05       0
  4978.0    0.05       0  5014.0    0.05       0
Bank Sta=4978,5014
Exp/Cntr=0.3,0.1

Type RM Length L Ch R = 1,541446,1910,1910,1910
BEGIN DESCRIPTION:
Mapping XS 58e1bcab
END DESCRIPTION:
XS GIS Cut Line= 3
      1560668.84      6909833.18      1560981.34      6906742.87
      1558221.67      6903792.27
#Sta/Elev= 30
  -640.1 1651.37    65.4 1643.32  1083.8 1642.91  1616.5 1634.49  2954.9 1640.01
  4787.2 1639.92  4886.4 1628.26  4992.4 1625.97  4995.4 1620.54  4996.0 1619.45
  4999.0 1618.05  5032.0 1619.45  5052.1 1628.78  5168.3 1638.42  5353.4 1642.74
  5495.0 1635.60  5629.4 1649.67  5749.6 1647.74  5777.9 1652.43  5848.7 1648.88
  5883.9 1656.92  5954.7 1657.14  6053.9 1673.42  6110.6 1676.90  6202.4 1661.00
  6287.4 1681.68  6336.7 1672.61  6372.4 1684.11  6492.6 1692.36  6506.0 1689.35
#Mann=6,-1,0
  -640.1    0.05       0  4995.4     0.1       0  4996.0    0.07       0
  5032.0     0.1       0  5052.1    0.12       0  5168.3    0.05       0
Bank Sta=4996,5032
Exp/Cntr=0.3,0.1

Type RM Length L Ch R = 1,539536,3364,3364,3364
BEGIN DESCRIPTION:
Mapping XS c7470c86
END DESCRIPTION:
XS GIS Cut Line= 3
      1560755.64      6909729.01      1561369.92      6906329.18
      1560078.24      6901933.30
#Sta/Elev= 30
  -478.3 1652.50   166.4 1642.83  1128.3 1642.99  1292.9 1638.98  1362.0 1642.81
  1433.2 1638.39  1778.7 1634.92  2243.5 1634.13  2276.6 1637.39  2360.7 1630.67
  2526.3 1636.58  2967.6 1634.30  4812.2 1637.73  4843.5 1637.53  4895.1 1630.17
  4937.3 1623.47  4968.6 1628.02  4979.0 1624.23  4980.6 1616.29  4983.6 1614.89
  5016.6 1616.29  5020.7 1621.77  5029.7 1625.97  5101.7 1637.33  5150.3 1638.68
  5777.4 1634.63  6630.4 1646.91  6907.2 1656.07  7450.0 1687.79  7558.3 1688.62
#Mann=5,-1,0
  -478.3    0.05       0  4895.1     0.1       0  4980.6    0.07       0
  5016.6     0.1       0  5150.3    0.05       0
Bank Sta=4980.6,5016.6
Exp/Cntr=0.3,0.1

Type RM Length L Ch R = 1,536172,634,634,634
BEGIN DESCRIPTION:
Mapping XS 9872ec2c
END DESCRIPTION:
XS GIS Cut Line= 5
      1561057.43      6908787.48      1561807.42      6907100.01
      1563099.08      6903975.01      1563453.25      6902725.01
      1564223.47      6900851.51
#Sta/Elev= 30
 -1098.7 1641.90  -473.4 1642.91   -38.4 1639.42   421.7 1642.21   580.8 1641.89
  1215.4 1640.63  1643.8 1633.40  2455.3 1631.68  4801.8 1636.42  4848.3 1627.64
  4885.0 1623.09  4980.1 1625.22  4987.5 1615.44  4990.5 1614.04  5023.5 1615.44
  5040.9 1624.78  5083.2 1634.01  5134.4 1637.39  5479.4 1632.19  5965.9 1633.04
  6161.2 1635.87  6225.4 1639.89  6238.5 1636.12  6571.4 1644.76  6737.0 1654.17
  6897.0 1654.72  7027.6 1663.05  7075.5 1660.90  7206.1 1669.71  7454.2 1671.96
#Mann=7,-1,0
 -1098.7    0.05       0   421.7   0.075       0   580.8    0.05       0
  4848.3     0.1       0  4987.5    0.07       0  5023.5     0.1       0
  5083.2    0.05       0
Bank Sta=4987.5,5023.5
Exp/Cntr=0.3,0.1

Type RM Length L Ch R = 1,535538,3492,3492,3492
BEGIN DESCRIPTION:
Mapping XS 37dc8d4d
END DESCRIPTION:
XS GIS Cut Line= 4
      1561828.24      6908787.55      1562619.92      6906683.35
      1563390.75      6904558.35      1564765.75      6901266.68
#Sta/Elev= 30
  -939.5 1640.95  -892.4 1642.32  -771.4 1642.00   143.0 1642.06   243.4 1643.05
   246.5 1643.15   453.6 1640.98   660.6 1641.60  1339.6 1631.91  2580.3 1633.58
  2837.4 1620.85  2893.3 1621.05  2918.6 1629.57  2979.8 1633.45  3830.9 1629.28
  4816.9 1634.30  4989.0 1624.19  4990.4 1612.24  4993.4 1610.84  5026.4 1612.24
  5054.3 1623.74  5118.9 1634.12  6057.3 1632.91  6181.4 1635.78  6257.2 1647.89
  6370.1 1646.54  6417.7 1660.41  6547.6 1658.58  6669.1 1670.14  7136.5 1668.10
#Mann=10,-1,0
  -939.5    0.05       0  -892.4   0.075       0  -771.4    0.05       0
   143.0     0.1       0   243.4   0.075       0   246.5     0.1       0
   453.6   0.075       0   660.6    0.05       0  4990.4    0.03       0
  5026.4    0.05       0
Bank Sta=4990.4,5026.4
Exp/Cntr=0.3,0.1

Type RM Length L Ch R = 1,532046,1825,1825,1825
BEGIN DESCRIPTION:
Mapping XS ef78b45c
END DESCRIPTION:
XS GIS Cut Line= 4
      1562099.07      6910454.20      1564369.92      6905516.68
      1565078.25      6903995.85      1565369.92      6901308.31
#Sta/Elev= 30
 -1294.3 1649.03  -140.0 1641.04   345.1 1641.84  1654.8 1640.29  1891.5 1640.08
  2154.2 1639.12  2159.6 1639.14  2671.3 1630.60  2721.3 1631.49  4580.2 1628.67
  4924.9 1631.99  4975.4 1612.60  4978.4 1611.20  5011.4 1612.60  5021.9 1621.14
  5032.5 1621.09  5136.1 1620.36  5400.9 1630.52  5679.0 1626.51  5753.1 1634.04
  6992.8 1629.05  7375.0 1636.01  7556.1 1647.23  7676.8 1652.35  7696.9 1647.51
  7776.5 1656.19  7998.7 1663.57  8129.4 1660.43  8148.0 1667.60  8521.4 1667.52
#Mann=14,-1,0
 -1294.3    0.05       0  -140.0   0.075       0   345.1    0.05       0
  1654.8   0.075       0  1891.5    0.05       0  2154.2    0.12       0
  2159.6    0.05       0  2671.3    0.12       0  2721.3    0.05       0
  4975.4    0.05       0  5011.4    0.05       0  5032.5     0.1       0
  5136.1    0.12       0  5400.9    0.05       0
Bank Sta=4975.4,5011.4
Exp/Cntr=0.3,0.1

Type RM Length L Ch R = 1,530221,843,843,843
BEGIN DESCRIPTION:
Mapping XS 8a25470f
END DESCRIPTION:
XS GIS Cut Line= 5
      1565040.45      6907127.53      1565630.73      6905512.94
      1566099.48      6903880.99      1566741.84      6901745.58
      1567019.62      6899783.72
#Sta/Elev= 30
  1747.4 1636.89  1853.4 1638.68  2077.0 1636.39  2492.2 1627.69  3152.3 1626.83
  3434.9 1630.93  4627.4 1631.56  4668.7 1625.33  4694.8 1621.42  4743.8 1619.67
  4969.9 1619.41  4977.5 1607.96  4981.3 1606.96  5022.5 1607.96  5024.3 1618.67
  5052.8 1631.54  5063.5 1631.69  5268.6 1628.66  7151.7 1625.18  7217.0 1622.03
  7349.1 1624.93  8351.4 1630.68  8482.7 1638.46  8525.3 1637.62  8553.4 1634.22
  8892.0 1643.39  9037.2 1652.15  9199.8 1662.86  9260.4 1669.35  9375.8 1668.48
#Mann=7,-1,0
  1747.4    0.05       0  4668.7    0.12       0  4743.8    0.05       0
  4977.5    0.05       0  5022.5    0.05       0  8892.0    0.12       0
  9037.2    0.05       0
Bank Sta=4977.5,5022.5
Exp/Cntr=0.3,0.1

Type RM Length L Ch R = 1,529378,2621,2621,2621
BEGIN DESCRIPTION:
Mapping XS f768a388
END DESCRIPTION:
XS GIS Cut Line= 5
      1563661.58      6911225.02      1565953.25      6905870.85
      1567001.40      6903810.36      1566911.58      6901641.68
      1567640.75      6899100.00
#Sta/Elev= 30
 -2363.2 1657.29 -1707.4 1640.43  -530.1 1639.38  -492.5 1639.65   427.7 1638.76
   673.0 1638.22  1984.6 1637.10  3459.6 1629.80  3621.1 1624.79  4362.5 1629.85
  4913.1 1619.98  4957.6 1617.17  4977.9 1607.46  4980.9 1606.06  5013.9 1607.46
  5034.7 1619.79  5079.6 1630.62  7816.7 1625.25  7906.7 1620.86  7942.4 1627.44
  8476.8 1624.25  9486.6 1635.61  9528.0 1644.03  9600.7 1640.87  9678.5 1645.38
  9705.1 1653.64  9757.1 1645.25  9857.6 1645.04 10114.6 1665.73 10587.3 1665.99
#Mann=7,-1,0
 -2363.2    0.05       0  -530.1   0.075       0  -492.5    0.05       0
   427.7   0.075       0   673.0    0.05       0  4977.9    0.03       0
  5013.9    0.05       0
Bank Sta=4977.9,5013.9
Exp/Cntr=0.3,0.1

Type RM Length L Ch R = 1,526757,2703,2703,2703
BEGIN DESCRIPTION:
Mapping XS 1039033d
END DESCRIPTION:
XS GIS Cut Line= 2
      1568932.42      6909537.51      1567953.25      6899183.31
#Sta/Elev= 30
   661.5 1644.06  1012.6 1638.60  2890.9 1638.82  3448.6 1634.28  4136.4 1632.76
  4186.7 1635.43  4668.8 1632.47  4789.3 1629.66  4919.9 1619.84  4960.1 1614.01
  4978.1 1606.52  4981.1 1605.12  5014.1 1606.52  5020.4 1616.10  5070.6 1619.38
  5111.9 1628.83  5152.1 1630.79  8676.6 1623.90  9287.5 1619.36  9460.1 1623.23
  9607.5 1616.65  9650.9 1620.39 10247.6 1631.85 10344.0 1636.46 10459.3 1648.78
 10504.7 1647.61 10621.0 1653.17 10765.0 1662.82 10796.0 1666.54 11061.9 1665.37
#Mann=6,-1,0
   661.5    0.05       0  4978.1    0.05       0  5014.1    0.05       0
  5111.9    0.05       0 10621.0    0.12       0 10765.0    0.05       0
Bank Sta=4978.1,5014.1
Exp/Cntr=0.3,0.1

Type RM Length L Ch R = 1,524054,3506,3506,3506
BEGIN DESCRIPTION:
Mapping XS d247e3b4
END DESCRIPTION:
XS GIS Cut Line= 3
      1570821.70      6906641.41      1569866.84      6904245.58
      1568234.88      6899523.32
#Sta/Elev= 30
  1666.8 1638.53  2183.2 1638.29  3159.2 1629.58  4124.4 1629.15  4538.3 1626.38
  4730.7 1629.16  4787.8 1626.80  4825.3 1618.97  4876.0 1613.25  4888.7 1615.59
  4933.3 1614.32  4962.8 1614.36  4982.0 1605.17  4985.0 1604.17  5018.0 1605.17
  5026.3 1617.86  5064.2 1622.90  5125.4 1628.82  6486.4 1621.61  8060.3 1621.04
  8185.1 1615.59  8210.9 1618.50  8616.3 1625.16  8829.2 1633.50  8948.6 1654.91
  9042.2 1654.70  9104.5 1648.90  9152.6 1653.66  9166.9 1651.64  9242.2 1653.12
#Mann=5,-1,0
  1666.8    0.05       0  4933.3     0.1       0  4982.0    0.07       0
  5018.0     0.1       0  5064.2    0.05       0
Bank Sta=4982,5018
Exp/Cntr=0.3,0.1

Type RM Length L Ch R = 1,520548,3893,3893,3893
BEGIN DESCRIPTION:
Clear Fork Brazos Rv 128.0
END DESCRIPTION:
XS GIS Cut Line= 3
      1571805.00      6907188.04      1571805.00      6902188.00
      1571305.00      6900187.99
#Sta/Elev= 30
     0.5 1647.23   350.5 1645.33   800.5 1636.09  1530.5 1629.14  2580.5 1628.69
  2930.5 1623.54  4130.5 1623.31  4590.5 1627.04  4720.5 1614.54  4840.5 1616.84
  4880.5 1613.00  4931.8 1614.48  4950.5 1611.50  4974.2 1601.47  4977.2 1600.07
  5010.2 1601.47  5010.8 1612.71  5052.1 1620.05  5059.8 1623.99  5103.2 1624.81
  6214.3 1617.95  6301.9 1616.47  6384.4 1611.89  6392.1 1609.66  6609.1 1619.13
  6763.2 1627.52  6841.4 1637.86  6948.7 1640.18  7020.9 1646.14  7062.1 1653.01
#Mann=7,-1,0
     0.5    0.05       0  4931.8    0.12       0  4974.2    0.07       0
  5010.2    0.12       0  5103.2    0.05       0  6609.1    0.12       0
  6841.4    0.05       0
Bank Sta=4974.2,5010.2
Exp/Cntr=0.3,0.1

Type RM Length L Ch R = 1,516655,2078,2078,2078
BEGIN DESCRIPTION:
Clear Fork Brazos Rv 127.0
END DESCRIPTION:
XS GIS Cut Line= 3
      1573704.99      6907288.04      1574705.00      6903788.00
      1572204.99      6899787.99
#Sta/Elev= 30
  1358.7 1646.28  1577.1 1644.71  1773.4 1639.07  1846.2 1632.98  2254.5 1629.86
  3811.9 1629.92  4885.4 1621.67  4915.6 1621.41  4942.9 1608.66  4957.2 1606.13
  4968.8 1598.30  4971.8 1596.90  5004.8 1598.30  5006.5 1610.45  5012.4 1610.95
  5173.9 1613.02  5222.8 1608.29  5252.9 1612.47  5383.8 1615.47  5446.2 1620.77
  8423.9 1617.14  8612.6 1615.76  8795.4 1609.01  8932.2 1616.78  9230.5 1624.76
  9303.0 1630.23  9352.0 1627.93  9382.6 1632.92  9577.2 1645.68  9715.8 1646.91
#Mann=5,-1,0
  1358.7    0.05       0  4885.4    0.12       0  4968.8    0.07       0
  5004.8    0.12       0  5446.2    0.05       0
Bank Sta=4968.8,5004.8
Exp/Cntr=0.3,0.1

Type RM Length L Ch R = 1,514577,3930,3930,3930
BEGIN DESCRIPTION:
Mapping XS 15226ee3
END DESCRIPTION:
XS GIS Cut Line= 3
      1577227.97      6904488.65      1576099.48      6903117.11
      1573095.98      6898933.04
#Sta/Elev= 30
  3491.6 1624.07  4475.1 1631.47  4524.6 1628.39  4808.7 1621.11  4905.5 1621.32
  4915.5 1621.02  4936.4 1611.46  4950.7 1604.76  4957.2 1596.33  4960.0 1596.23
  4963.8 1595.23  5005.0 1596.23  5007.6 1608.18  5014.6 1610.05  5028.9 1609.87
  5049.7 1605.16  5064.1 1609.01  5082.3 1609.53  5121.4 1611.38  5163.1 1620.54
  5191.8 1620.78  7800.5 1616.30  8817.3 1617.43  9362.4 1614.69  9504.9 1607.54
  9605.6 1613.58  9907.4 1620.81 10085.7 1628.97 10136.0 1628.41 10418.2 1634.75
#Mann=5,-1,0
  3491.6    0.05       0  4905.5     0.1       0  4960.0    0.07       0
  5005.0     0.1       0  5082.3    0.05       0
Bank Sta=4960,5005
Exp/Cntr=0.3,0.1

Type RM Length L Ch R = 1,510647,3714,3714,3714
BEGIN DESCRIPTION:
Mapping XS 48af7542
END DESCRIPTION:
XS GIS Cut Line= 3
      1578557.40      6904641.64      1577619.92      6901850.01
      1575932.40      6897579.15
#Sta/Elev= 30
  1566.3 1623.57  3490.0 1625.73  3910.4 1618.02  4207.3 1616.19  4958.6 1618.80
  4964.9 1617.71  4986.4 1604.86  4989.5 1594.03  4992.5 1592.63  5025.5 1594.03
  5026.0 1601.29  5031.4 1604.24  5065.0 1605.68  5109.8 1606.82  5134.2 1615.65
  5171.4 1619.40  6706.8 1611.09  7146.4 1609.70  7190.6 1612.26  7230.2 1609.63
  7235.6 1605.45  7289.7 1602.24  7362.7 1605.44  7368.1 1607.93  7405.7 1611.50
  7722.4 1612.80  7825.0 1615.79  8416.4 1623.94  8685.2 1622.26  9103.3 1623.97
#Mann=6,-1,0
  1566.3    0.05       0  4958.6     0.1       0  4989.5    0.07       0
  5025.5     0.1       0  5065.0    0.12       0  5171.4    0.05       0
Bank Sta=4989.5,5025.5
Exp/Cntr=0.3,0.1

Type RM Length L Ch R = 1,506933,4100,4100,4100
BEGIN DESCRIPTION:
Mapping XS afa7b18e
END DESCRIPTION:
XS GIS Cut Line= 5
      1581255.72      6902960.83      1580960.59      6901693.49
      1580769.62      6901467.80      1579589.06      6900946.97
      1576342.54      6897440.03
#Sta/Elev= 30
  3513.1 1619.41  4512.7 1620.18  4532.5 1618.35  4829.4 1615.05  4964.6 1615.83
  4971.1 1609.74  4982.0 1594.27  4985.0 1593.27  5018.0 1594.27  5020.5 1598.17
  5034.8 1603.37  5342.0 1604.41  5394.1 1606.25  5446.2 1604.98  5539.4 1609.26
  5585.0 1615.80  5614.9 1616.69  5690.3 1613.40  5902.0 1617.28  7654.8 1612.16
  8801.2 1611.46  8957.2 1610.22  9070.0 1607.00  9134.0 1602.80  9176.6 1602.75
  9317.8 1611.12  9516.2 1610.43  9820.1 1617.54 10167.1 1617.40 11179.3 1623.50
#Mann=3,-1,0
  3513.1    0.05       0  4982.0    0.05       0  5018.0    0.05       0
Bank Sta=4982,5018
Exp/Cntr=0.3,0.1

Type RM Length L Ch R = 1,502833,3124,3124,3124
BEGIN DESCRIPTION:
Mapping XS 7ae39abf
END DESCRIPTION:
XS GIS Cut Line= 3
      1581554.27      6903010.24      1580165.37      6898947.73
      1576502.17      6896048.42
#Sta/Elev= 30
  1592.6 1619.30  2688.2 1619.46  2704.6 1617.76  2719.6 1618.73  3106.2 1614.59
  3529.0 1616.12  4807.7 1613.39  4916.0 1614.70  4947.3 1609.85  4973.4 1600.56
  4978.7 1601.65  4981.2 1590.22  4984.2 1588.82  5014.2 1588.82  5017.2 1590.22
  5036.0 1600.10  5098.6 1602.54  5114.2 1600.92  5129.9 1601.77  5155.9 1611.02
  5161.2 1610.83  5167.0 1613.91  5198.7 1615.22  7330.8 1608.04  7380.5 1606.46
  8149.8 1610.95  8911.0 1610.04  9345.4 1612.10  9851.9 1621.36 10557.7 1624.92
#Mann=3,-1,0
  1592.6    0.05       0  4981.2    0.05       0  5017.2    0.05       0
Bank Sta=4981.2,5017.2
Exp/Cntr=0.3,0.1

Type RM Length L Ch R = 1,499709,3999,3999,3999
BEGIN DESCRIPTION:
Mapping XS ec7414e6
END DESCRIPTION:
XS GIS Cut Line= 5
      1582280.04      6902874.08      1581724.48      6901016.41
      1581672.40      6900009.47      1580127.26      6894974.74
      1578808.91      6894315.57
#Sta/Elev= 30
  3398.3 1617.77  4763.2 1615.47  4907.7 1599.86  4972.3 1599.15  4980.7 1593.31
  4982.0 1588.87  4985.0 1587.87  5018.0 1588.87  5022.5 1597.95  5038.5 1601.61
  5214.4 1601.88  5247.5 1613.03  5293.9 1614.34  7513.0 1611.79  8803.9 1603.37
  9288.3 1606.84  9386.5 1603.29  9527.9 1607.19  9724.3 1603.23 10217.4 1608.67
 10344.9 1604.10 10481.0 1608.73 11791.3 1610.21 11849.4 1596.93 11886.4 1604.03
 11908.7 1604.13 11938.8 1598.11 11961.2 1606.38 12037.3 1610.82 13086.0 1612.26
#Mann=3,-1,0
  3398.3    0.05       0  4982.0    0.05       0  5018.0    0.05       0
Bank Sta=4982,5018
Exp/Cntr=0.3,0.1

Type RM Length L Ch R = 1,495710,1816,1816,1816
BEGIN DESCRIPTION:
Mapping XS 32d1820f
END DESCRIPTION:
XS GIS Cut Line= 4
      1582883.81      6903468.06      1583238.29      6902333.15
      1583161.58      6899391.68      1581786.77      6894142.38
#Sta/Elev= 30
   -80.6 1617.85  3454.3 1607.33  4851.1 1610.32  4974.7 1594.70  4983.0 1585.15
  4986.0 1583.75  5019.0 1585.15  5026.4 1597.84  5067.7 1607.72  5140.1 1609.32
  5714.3 1605.64  5795.1 1601.20  5830.4 1605.56  5863.7 1602.32  6556.3 1606.49
  6732.0 1604.13  8851.2 1608.69  8975.2 1604.87  8985.5 1603.54  8995.9 1595.89
  9006.2 1595.72  9016.6 1600.37  9066.4 1604.24  9119.9 1600.43  9202.6 1604.68
  9233.6 1610.79  9263.3 1610.15  9295.7 1616.44  9368.0 1641.02  9477.2 1645.53
#Mann=3,-1,0
   -80.6    0.05       0  4983.0    0.05       0  5019.0    0.05       0
Bank Sta=4983,5019
Exp/Cntr=0.3,0.1

Type RM Length L Ch R = 1,493894,419,419,419
BEGIN DESCRIPTION:
Mapping XS 1bf80fd8
END DESCRIPTION:
XS GIS Cut Line= 6
      1583407.12      6901860.01      1583900.36      6899687.06
      1584780.21      6898833.87      1586206.63      6897020.85
      1586593.23      6896460.95      1586766.54      6895647.75
#Sta/Elev= 30
  2199.9 1612.64  4686.7 1606.80  4794.1 1599.92  4829.3 1607.27  4950.8 1608.34
  4971.9 1588.65  4982.0 1584.70  4985.0 1583.70  5018.0 1584.70  5021.5 1598.17
  5092.0 1595.18  5164.1 1600.73  5192.3 1607.46  5258.6 1608.49  7991.9 1602.56
  8186.4 1589.53  8258.5 1598.45  8285.6 1593.34  8315.3 1595.18  8321.4 1590.21
  8351.1 1587.61  8366.0 1597.20  8380.8 1600.07  8443.8 1587.42  8479.6 1591.52
  8560.0 1584.70  8687.3 1600.10  8781.2 1594.43  8874.5 1601.91  9488.2 1624.61
#Mann=3,-1,0
  2199.9    0.05       0  4982.0    0.03       0  5018.0    0.05       0
Bank Sta=4982,5018
Exp/Cntr=0.3,0.1

Type RM Length L Ch R = 1,493475,11325,11325,11325
BEGIN DESCRIPTION:
Mapping XS d45f5f49
END DESCRIPTION:
XS GIS Cut Line= 6
      1583647.07      6901886.69      1584273.63      6899780.38
      1584980.18      6899153.82      1586193.30      6897340.80
      1586953.17      6895981.03      1586926.51      6895714.41
#Sta/Elev= 30
  2423.6 1612.69  4808.2 1607.94  4978.0 1595.49  4982.0 1583.56  4985.0 1582.56
  5018.0 1583.56  5049.1 1594.07  5131.5 1602.11  5162.0 1608.88  5225.3 1608.96
  7439.4 1600.99  7526.4 1596.96  7577.5 1601.89  8130.6 1603.06  8290.5 1592.99
  8349.1 1597.41  8400.6 1593.27  8451.0 1597.40  8467.3 1593.64  8516.8 1601.32
  8605.4 1602.62  8650.7 1601.41  8763.2 1583.56  8785.1 1588.63  8790.8 1585.35
  8807.0 1591.95  8894.8 1596.17  8976.9 1593.40  9026.5 1602.89  9572.9 1622.51
#Mann=5,-1,0
  2423.6    0.05       0  4982.0    0.05       0  5018.0    0.05       0
  5131.5    0.12       0  5225.3    0.05       0
Bank Sta=4982,5018
Exp/Cntr=0.3,0.1

Type RM Length L Ch R = 1,482150,3837,3837,3837
BEGIN DESCRIPTION:
Clear Fork Brazos Rv 123.0
END DESCRIPTION:
XS GIS Cut Line= 3
      1587004.99      6907038.04      1589005.00      6897038.00
      1589005.00      6896537.98
#Sta/Elev= 30
 -5192.1 1637.13 -4722.9 1634.72 -4692.4 1637.19 -4610.8 1633.65 -4580.2 1629.46
 -4549.6 1632.03 -4417.0 1624.75 -4264.0 1619.71 -3917.3 1614.72   182.3 1607.23
   559.6 1601.01  4281.9 1599.72  4751.0 1603.71  4781.6 1601.75  4812.2 1594.01
  4873.4 1588.17  4883.6 1584.34  4893.8 1584.21  4914.6 1590.58  4965.2 1588.97
  4980.2 1579.51  4983.2 1577.81  5016.2 1579.51  5026.0 1590.38  5066.0 1600.81
  5082.1 1601.89  5126.0 1603.16  5166.0 1608.40  5286.0 1613.07  5506.0 1614.74
#Mann=5,-1,0
 -5192.1    0.05       0  4914.6     0.1       0  4980.2    0.07       0
  5016.2     0.1       0  5082.1    0.05       0
Bank Sta=4980.2,5016.2
Exp/Cntr=0.3,0.1

Type RM Length L Ch R = 1,478313,3829,3829,3829
BEGIN DESCRIPTION:
Clear Fork Brazos Rv 122.0
END DESCRIPTION:
XS GIS Cut Line= 4
      1587439.68      6906742.88      1588355.00      6901988.00
      1590855.00      6899488.00      1593355.01      6897987.99
#Sta/Elev= 30
 -3378.3 1637.08 -2915.1 1633.44 -2583.6 1617.27 -2318.9 1614.10  1392.6 1609.43
  1845.7 1599.06  4674.1 1598.58  4858.0 1595.51  4900.4 1589.57  4914.6 1592.45
  4971.1 1584.96  4980.4 1577.37  4983.4 1575.67  5016.4 1577.37  5057.7 1589.00
  5129.6 1584.46  5357.0 1589.91  5442.6 1600.29  6452.7 1598.27  6682.6 1594.94
  7022.5 1608.10  7170.5 1613.21  7207.4 1620.73  7324.0 1609.90  7530.0 1618.68
  7646.7 1616.51  7716.6 1626.38  7753.6 1623.22  7798.3 1630.96  7914.9 1634.76
#Mann=5,-1,0
 -3378.3    0.05       0  4980.4    0.05       0  5016.4    0.05       0
  6452.7    0.12       0  7022.5    0.05       0
Bank Sta=4980.4,5016.4
Exp/Cntr=0.3,0.1
