HEC-RAS study Clear Fork Brazos Rv.prj: Clear Fork Brazos Rv Base Level Engineering

--- Clear Fork Brazos Rv.g01 (geometry) --- (continued)

Type RM Length L Ch R = 1,339612,2152,2152,2152
BEGIN DESCRIPTION:
Mapping XS 8e5bb11e
END DESCRIPTION:
XS GIS Cut Line= 4
      1632937.22      6984792.91      1632752.25      6984003.68
      1633085.22      6981228.90      1633380.87      6979541.20
#Sta/Elev= 30
  4274.9 1525.04  4362.1 1524.65  4495.6 1518.65  4649.7 1515.99  4803.8 1506.66
  4855.1 1506.93  4921.0 1496.35  4937.3 1484.95  4957.8 1478.21  4973.0 1469.51
  4977.5 1468.51  5027.0 1469.51  5040.0 1471.65  5048.3 1482.56  5085.5 1487.63
  5117.9 1500.34  5148.6 1504.56  5216.2 1504.84  5312.8 1503.70  5433.7 1497.51
  5909.0 1502.20  6998.5 1503.30  7266.7 1508.14  7861.0 1513.28  8080.4 1511.63
  8642.5 1513.19  9058.8 1518.50  9343.0 1525.42  9485.2 1531.67  9593.6 1541.30
#Mann=5,-1,0
  4274.9    0.05       0  4973.0    0.05       0  5027.0    0.05       0
  5117.9    0.12       0  5216.2    0.05       0
#XS Ineff=2,0
       0                 5164.40    0.00 1512.80
Permanent Ineff=
       F       F
Bank Sta=4973,5027
Exp/Cntr=0.3,0.1

Type RM Length L Ch R = 1,337460,2340,2340,2340
BEGIN DESCRIPTION:
Mapping XS 866e5e92
END DESCRIPTION:
XS GIS Cut Line= 3
      1634956.69      6984140.06      1633229.49      6981205.89
      1633538.69      6979321.98
#Sta/Elev= 30
  3644.4 1514.40  3916.7 1514.11  4188.1 1507.87  4231.0 1509.88  4481.0 1503.07
  4732.7 1502.39  4779.7 1503.50  4830.4 1494.16  4859.7 1495.07  4888.4 1490.90
  4918.3 1481.13  4924.1 1471.44  4927.1 1470.84  4936.1 1469.46  4942.9 1468.46
  5017.1 1469.46  5035.5 1480.08  5056.9 1485.97  5115.5 1497.11  5174.1 1501.35
  5861.4 1500.07  6421.6 1510.20  7634.8 1511.77  8104.0 1516.46  8476.7 1527.40
  8638.1 1538.00  8739.4 1551.33  8800.2 1552.46  8839.3 1558.50  8958.3 1561.59
#Mann=5,-1,0
  3644.4    0.05       0  4732.7    0.12       0  4927.1    0.05       0
  4936.1    0.03       0  5017.1    0.05       0
Bank Sta=4936.1,5017.1
Exp/Cntr=0.3,0.1

Type RM Length L Ch R = 1,335120,3186,3186,3186
BEGIN DESCRIPTION:
Mapping XS ea6ca10d
END DESCRIPTION:
XS GIS Cut Line= 2
      1635477.54      6984487.32      1635293.13      6980321.80
#Sta/Elev= 30
  1547.6 1514.81  1727.1 1513.94  2187.5 1505.23  3068.4 1499.91  4619.9 1502.79
  4656.2 1499.36  4661.2 1500.98  4701.9 1495.25  4733.7 1498.29  4766.2 1492.42
  4890.2 1475.43  4980.3 1471.76  4987.7 1469.00  4991.4 1468.00  5032.7 1469.00
  5040.3 1471.43  5050.3 1480.41  5060.4 1482.62  5070.4 1488.93  5090.4 1493.18
  5107.6 1501.78  5129.4 1501.39  5190.5 1503.26  5240.5 1515.61  5290.6 1536.32
  5326.9 1540.70  5400.7 1543.14  5470.8 1557.92  5500.8 1561.17  5717.2 1569.69
#Mann=8,-1,0
  1547.6    0.05       0  4701.9    0.12       0  4733.7    0.05       0
  4766.2    0.12       0  4987.7    0.07       0  5032.7    0.12       0
  5129.4    0.12       0  5326.9    0.05       0
Bank Sta=4987.7,5032.7
Exp/Cntr=0.3,0.1

Type RM Length L Ch R = 1,331934,4735,4735,4735
BEGIN DESCRIPTION:
Mapping XS 62725a57
END DESCRIPTION:
XS GIS Cut Line= 2
      1635662.03      6984693.46      1638297.82      6982372.23
#Sta/Elev= 30
  2025.2 1515.70  3327.7 1501.90  3887.5 1498.19  4369.4 1500.23  4759.3 1493.46
  4879.8 1496.02  4900.7 1494.36  4921.6 1485.76  4935.8 1483.56  4943.4 1480.44
  4950.1 1466.78  4952.6 1466.78  4960.1 1465.78  5042.6 1466.78  5056.3 1478.03
  5063.9 1476.41  5070.6 1481.19  5078.1 1479.41  5084.8 1482.38  5092.1 1480.62
  5099.0 1480.93  5141.7 1495.25  5205.3 1490.79  5219.5 1492.81  5333.3 1519.94
  5360.9 1537.15  5375.1 1541.02  5446.2 1553.41  5516.2 1560.17  5537.4 1562.19
#Mann=5,-1,0
  2025.2    0.05       0  4952.6    0.03       0  5042.6    0.05       0
  5092.1    0.12       0  5516.2    0.05       0
Bank Sta=4952.6,5042.6
Exp/Cntr=0.3,0.1

Type RM Length L Ch R = 1,327199,3304,3304,3304
BEGIN DESCRIPTION:
Clear Fork Brazos Rv 84.0
END DESCRIPTION:
XS GIS Cut Line= 3
      1640797.68      6985854.78      1641014.69      6985533.60
      1641705.00      6983187.99
#Sta/Elev= 30
  4147.6 1555.60  4489.4 1533.10  4603.6 1500.22  4655.4 1489.39  4780.8 1478.99
  4926.7 1478.64  4958.0 1470.89  4975.0 1462.85  4978.7 1461.85  5020.0 1462.85
  5041.4 1467.66  5062.3 1467.56  5112.6 1483.51  5135.2 1491.42  5153.5 1492.50
  5313.4 1494.28  5507.8 1498.44  6011.1 1491.80  6123.0 1482.00  6144.5 1480.89
  6156.8 1487.73  6288.3 1490.02  6326.9 1487.30  6448.7 1496.13  6479.9 1508.29
  6532.1 1513.05  6676.0 1561.39  6730.3 1569.42  6819.8 1581.56  6980.3 1586.95
#Mann=7,-1,0
  4147.6    0.05       0  4975.0    0.05       0  5020.0    0.05       0
  5112.6    0.12       0  5313.4    0.05       0  6123.0    0.12       0
  6730.3    0.05       0
#XS Ineff=2,0
       0                 5480.90    0.00 1506.61
Permanent Ineff=
       F       F
Bank Sta=4975,5020
Exp/Cntr=0.3,0.1

Type RM Length L Ch R = 1,323895,1918,1918,1918
BEGIN DESCRIPTION:
Mapping XS b8737ab3
END DESCRIPTION:
XS GIS Cut Line= 2
      1642400.30      6987395.30      1644660.28      6985820.23
#Sta/Elev= 30
  3148.7 1515.72  3344.2 1516.11  3710.7 1499.82  4026.6 1498.08  4277.0 1487.03
  4342.4 1489.91  4420.1 1488.36  4544.6 1491.51  4598.7 1492.52  4744.7 1490.99
  4759.5 1485.93  4795.3 1481.65  4902.6 1473.19  4946.2 1466.94  4971.9 1459.98
  4976.4 1458.98  5025.9 1459.98  5054.4 1475.71  5068.1 1478.18  5182.7 1485.10
  5218.5 1492.46  5290.0 1513.13  5319.7 1525.79  5361.6 1538.60  5406.1 1566.24
  5447.9 1579.29  5456.7 1585.03  5477.6 1590.56  5533.1 1591.43  5903.4 1598.10
#Mann=7,-1,0
  3148.7    0.05       0  4420.1    0.12       0  4544.6    0.05       0
  4598.7    0.12       0  4971.9    0.07       0  5025.9    0.12       0
  5533.1    0.05       0
Bank Sta=4971.9,5025.9
Exp/Cntr=0.3,0.1

Type RM Length L Ch R = 1,321977,3764,3764,3764
BEGIN DESCRIPTION:
Mapping XS 1de1d8a1
END DESCRIPTION:
XS GIS Cut Line= 2
      1642519.61      6987861.87      1644885.09      6988404.41
#Sta/Elev= 30
  3520.5 1511.63  3587.6 1510.52  3895.4 1518.16  4379.1 1491.90  4531.5 1488.19
  4823.3 1489.53  4864.2 1486.15  4900.8 1479.02  4962.4 1474.77  4972.6 1471.47
  4982.3 1459.96  4988.3 1458.96  5054.3 1459.96  5090.8 1471.94  5138.9 1476.81
  5207.6 1491.39  5224.7 1498.68  5259.9 1506.00  5280.4 1516.46  5310.5 1519.78
  5321.5 1518.13  5358.5 1528.28  5363.6 1526.79  5444.2 1542.85  5465.1 1544.01
  5535.1 1558.70  5759.8 1579.96  5824.2 1582.13  5893.6 1590.29  5947.4 1592.41
#Mann=6,-1,0
  3520.5    0.05       0  4864.2     0.1       0  4982.3    0.07       0
  5054.3     0.1       0  5090.8    0.12       0  5207.6    0.05       0
Bank Sta=4982.3,5054.3
Exp/Cntr=0.3,0.1

Type RM Length L Ch R = 1,318213,3310,3310,3310
BEGIN DESCRIPTION:
Mapping XS 5729e91d
END DESCRIPTION:
XS GIS Cut Line= 2
      1641879.42      6991355.80      1645720.27      6991475.15
#Sta/Elev= 30
  4076.9 1588.30  4232.6 1589.55  4402.6 1583.79  4492.7 1577.45  4542.7 1555.66
  4592.7 1526.34  4629.1 1514.95  4634.1 1517.03  4702.8 1495.97  4772.8 1483.68
  4832.8 1479.83  4852.9 1475.01  4882.9 1459.93  4902.9 1462.36  4991.7 1460.03
  4995.2 1457.34  4998.2 1456.34  5031.2 1457.34  5042.9 1458.81  5063.0 1471.46
  5353.1 1485.84  6080.8 1485.91  6424.7 1492.76  6773.8 1497.64  7043.9 1506.15
  7523.7 1533.03  7724.2 1572.30  7774.3 1578.95  7864.3 1583.98  7919.6 1583.21
#Mann=7,-1,0
  4076.9    0.05       0  4991.7    0.12       0  4995.2    0.07       0
  5031.2    0.12       0  6080.8    0.05       0  6424.7    0.12       0
  6773.8    0.05       0
Bank Sta=4995.2,5031.2
Exp/Cntr=0.3,0.1

Type RM Length L Ch R = 1,314903,2180,2180,2180
BEGIN DESCRIPTION:
Mapping XS 17d3d0be
END DESCRIPTION:
XS GIS Cut Line= 3
      1642063.89      6994524.21      1643224.94      6994318.05
      1645264.84      6993959.98
#Sta/Elev= 30
  2863.3 1552.74  2982.9 1518.10  3036.9 1508.79  3219.9 1496.47  3433.2 1491.11
  4421.0 1491.57  4731.9 1483.77  4885.9 1473.83  4934.0 1461.85  4949.8 1456.37
  4967.8 1452.69  4970.8 1451.69  5003.8 1452.69  5017.2 1462.57  5053.9 1470.79
  5136.2 1471.21  5271.1 1468.13  5332.0 1462.13  5352.3 1455.66  5382.8 1464.13
  5392.9 1459.42  5413.2 1467.67  5484.1 1480.05  5495.0 1482.88  5578.1 1485.02
  5751.2 1499.33  5805.5 1511.77  5869.5 1519.90  6045.7 1556.61  6113.6 1575.48
#Mann=11,-1,0
  2863.3    0.05       0  4731.9    0.12       0  4934.0    0.05       0
  4949.8    0.12       0  4967.8    0.07       0  5003.8    0.12       0
  5136.2    0.05       0  5484.1    0.12       0  5495.0    0.05       0
  5869.5    0.12       0  6045.7    0.05       0
Bank Sta=4967.8,5003.8
Exp/Cntr=0.3,0.1

Type RM Length L Ch R = 1,312723,2319,2319,2319
BEGIN DESCRIPTION:
Clear Fork Brazos Rv 80.0
END DESCRIPTION:
XS GIS Cut Line= 3
      1642212.62      6995177.71      1644205.00      6995938.00
      1644641.54      6996088.60
#Sta/Elev= 30
  2862.4 1500.73  2879.1 1500.62  2918.5 1493.98  3133.8 1489.26  3903.2 1488.61
  4555.4 1491.39  4698.7 1485.47  4730.6 1484.28  4810.1 1475.29  4815.5 1472.92
  4840.2 1473.59  4887.9 1466.83  4941.4 1470.16  4979.9 1459.03  4984.4 1451.69
  4990.4 1450.69  5056.4 1451.69  5067.6 1452.52  5072.9 1461.45  5079.5 1464.02
  5090.1 1465.64  5130.0 1479.75  5248.8 1479.74  5317.2 1484.59  5348.4 1493.61
  5354.6 1497.38  5379.6 1502.57  5428.6 1521.44  5442.0 1528.01  5456.7 1542.17
#Mann=4,-1,0
  2862.4    0.05       0  4698.7    0.12       0  4984.4    0.07       0
  5056.4    0.12       0
Bank Sta=4984.4,5056.4
Exp/Cntr=0.3,0.1

Type RM Length L Ch R = 1,310404,2015,2015,2015
BEGIN DESCRIPTION:
Mapping XS 676dc003
END DESCRIPTION:
XS GIS Cut Line= 3
      1641944.58      6996846.27      1644223.20      6998311.10
      1644950.09      6998180.91
#Sta/Elev= 30
  3118.5 1530.99  3221.7 1501.91  3279.2 1494.50  3309.2 1485.87  3351.8 1491.68
  4350.4 1482.97  4828.6 1483.36  4849.7 1476.95  4864.9 1474.04  4870.9 1476.55
  4886.1 1471.20  4928.3 1462.38  4943.5 1462.24  4973.8 1454.38  4982.5 1450.95
  4985.5 1449.95  5018.5 1450.95  5031.4 1456.21  5052.5 1458.62  5080.5 1458.89
  5146.3 1452.50  5182.6 1458.44  5188.5 1463.03  5203.7 1467.32  5230.5 1469.17
  5297.5 1469.30  5364.2 1480.17  5442.8 1480.69  6104.4 1501.21  6565.8 1528.73
#Mann=5,-1,0
  3118.5    0.05       0  4973.8    0.12       0  4982.5    0.07       0
  5018.5    0.12       0  5230.5    0.05       0
Bank Sta=4982.5,5018.5
Exp/Cntr=0.3,0.1

Type RM Length L Ch R = 1,308389,982,982,982
BEGIN DESCRIPTION:
Mapping XS c0a6bf55
END DESCRIPTION:
XS GIS Cut Line= 3
      1640812.59      6999070.86      1643407.79      6999684.78
      1644784.47      6998429.02
#Sta/Elev= 30
  3212.1 1565.94  3310.2 1560.49  3512.6 1538.41  3651.1 1500.57  3738.1 1484.00
  3952.7 1475.05  4260.8 1480.76  4435.0 1477.63  4482.4 1472.45  4519.5 1475.49
  4540.2 1471.76  4560.7 1477.13  4609.2 1478.26  4663.5 1462.61  4848.5 1479.51
  4909.3 1476.66  4940.9 1475.85  4957.7 1454.19  4974.2 1450.06  4978.7 1449.06
  5028.2 1450.06  5095.1 1459.95  5137.0 1457.18  5174.2 1464.49  5280.1 1464.58
  5351.3 1472.74  5413.6 1479.58  6079.7 1487.80  7035.7 1486.99  7742.3 1511.99
#Mann=7,-1,0
  3212.1    0.05       0  3651.1    0.12       0  3952.7    0.05       0
  4909.3    0.12       0  4974.2    0.07       0  5028.2    0.12       0
  5351.3    0.05       0
Bank Sta=4974.2,5028.2
Exp/Cntr=0.3,0.1

Type RM Length L Ch R = 1,307407,2269,2269,2269
BEGIN DESCRIPTION:
Mapping XS d23fb629
END DESCRIPTION:
XS GIS Cut Line= 4
      1641621.83      7001014.97      1641769.90      7000577.01
      1643106.70      7000186.38      1644885.13      6998506.38
#Sta/Elev= 30
  3927.5 1541.50  3951.9 1537.18  3955.6 1538.58  4008.8 1533.17  4020.0 1530.38
  4046.2 1516.10  4061.5 1513.18  4077.6 1506.20  4146.0 1487.57  4177.7 1480.89
  4209.3 1477.88  4323.9 1474.60  4834.9 1481.08  4868.4 1477.06  4895.2 1467.63
  4916.0 1464.14  4943.7 1449.57  4950.4 1448.57  5024.7 1449.57  5030.6 1455.85
  5051.5 1461.73  5092.4 1463.59  5151.6 1477.62  5395.2 1480.52  5762.0 1477.57
  6112.5 1480.83  6424.0 1487.40  7407.1 1486.50  7753.8 1494.76  8229.0 1513.46
#Mann=6,-1,0
  3927.5    0.12       0  3955.6    0.05       0  4943.7    0.05       0
  5024.7    0.05       0  5092.4    0.12       0  5395.2    0.05       0
Bank Sta=4943.7,5024.7
Exp/Cntr=0.3,0.1

Type RM Length L Ch R = 1,305138,2183,2183,2183
BEGIN DESCRIPTION:
Mapping XS 0c69a64c
END DESCRIPTION:
XS GIS Cut Line= 2
      1643984.50      7002054.57      1645047.86      6998538.97
#Sta/Elev= 30
  4459.7 1571.90  4529.2 1570.45  4551.6 1567.67  4571.0 1562.26  4602.4 1559.49
  4650.4 1529.77  4665.1 1525.91  4683.3 1513.27  4706.9 1504.82  4721.5 1502.89
  4754.5 1491.00  4825.6 1475.99  4858.5 1465.35  4915.8 1461.26  4936.7 1462.49
  4947.1 1458.67  4957.3 1449.15  4962.3 1449.15  4969.8 1448.15  5052.3 1449.15
  5072.5 1460.73  5091.1 1463.82  5132.5 1476.23  5267.8 1473.47  5574.0 1483.31
  6462.0 1482.06  7307.0 1490.82  7898.4 1510.42  8029.1 1512.04  8132.6 1517.51
#Mann=5,-1,0
  4459.7    0.05       0  4962.3    0.03       0  5052.3    0.05       0
  5091.1    0.12       0  5267.8    0.05       0
Bank Sta=4962.3,5052.3
Exp/Cntr=0.3,0.1

Type RM Length L Ch R = 1,302955,1814,1814,1814
BEGIN DESCRIPTION:
Mapping XS 477dd2df
END DESCRIPTION:
XS GIS Cut Line= 3
      1646447.59      7001696.51      1645807.41      7000492.09
      1645850.76      6999451.69
#Sta/Elev= 30
  4540.5 1572.28  4578.2 1561.08  4584.1 1555.69  4606.8 1547.34  4622.2 1544.25
  4638.5 1535.58  4666.1 1526.52  4748.4 1490.83  4808.7 1475.08  4844.6 1471.83
  4867.2 1474.42  4896.6 1473.72  4940.5 1456.13  4946.5 1449.12  4952.2 1449.12
  4960.4 1448.12  5051.2 1449.12  5066.7 1458.99  5090.5 1461.87  5105.0 1465.81
  5116.4 1466.07  5198.6 1463.50  5319.1 1464.71  5368.8 1469.80  5459.9 1475.47
  5546.7 1479.27  5829.6 1477.91  6008.7 1479.33  6450.7 1495.47  6945.8 1502.75
#Mann=5,-1,0
  4540.5    0.05       0  4952.2    0.03       0  5051.2    0.05       0
  5090.5    0.12       0  5459.9    0.05       0
Bank Sta=4952.2,5051.2
Exp/Cntr=0.3,0.1

Type RM Length L Ch R = 1,301141,1141,1141,1141
BEGIN DESCRIPTION:
Clear Fork Brazos Rv 77.0
END DESCRIPTION:
XS GIS Cut Line= 3
      1648054.97      7000687.97      1647555.00      7000188.00
      1647054.98      6999687.98
#Sta/Elev= 30
  4292.7 1584.90  4391.7 1579.39  4419.9 1574.24  4434.1 1567.27  4448.2 1557.71
  4476.5 1541.58  4528.6 1520.36  4617.9 1494.60  4664.8 1478.86  4664.9 1478.82
  4688.6 1470.26  4716.9 1466.00  4801.8 1460.03  4858.3 1459.23  4886.6 1456.08
  4914.9 1455.68  4919.2 1453.44  4927.5 1449.11  4935.8 1448.11  5026.5 1449.11
  5042.2 1455.71  5056.3 1468.17  5070.5 1473.26  5084.6 1474.41  5112.9 1475.82
  5183.6 1473.69  5240.2 1474.04  5381.6 1481.21  5537.2 1485.07  5706.9 1492.35
#Mann=7,-1,0
  4292.7    0.05       0  4528.6    0.12       0  4664.8    0.05       0
  4664.9    0.12       0  4919.2    0.05       0  4927.5    0.03       0
  5026.5    0.05       0
Bank Sta=4927.5,5026.5
Exp/Cntr=0.3,0.1

Type RM Length L Ch R = 1,300000,2384,2384,2384
BEGIN DESCRIPTION:
Mapping XS 53526ef3
END DESCRIPTION:
XS GIS Cut Line= 2
      1648704.52      6999602.32      1646935.90      6998549.83
#Sta/Elev= 30
  4586.4 1552.01  4641.0 1551.83  4678.0 1544.86  4855.6 1492.14  4896.1 1473.89
  4924.7 1464.07  4954.5 1455.81  4969.9 1449.28  4977.1 1449.10  4986.1 1448.10
  5085.1 1449.10  5092.8 1457.02  5098.6 1459.46  5129.8 1460.81  5144.4 1464.05
  5151.5 1467.87  5179.3 1473.62  5256.4 1473.83  5264.9 1473.64  5406.3 1470.72
  5493.5 1478.92  5538.1 1478.87  5691.3 1478.65  5741.2 1480.90  6063.7 1504.09
  6296.4 1506.55  6354.6 1508.15  6377.9 1510.80  6420.9 1507.58  6644.5 1510.15
#Mann=9,-1,0
  4586.4    0.05       0  4855.6    0.12       0  4924.7    0.05       0
  4977.1    0.03       0  5085.1    0.05       0  5151.5    0.12       0
  5256.4    0.05       0  5264.9    0.12       0  5538.1    0.05       0
Bank Sta=4977.1,5085.1
Exp/Cntr=0.3,0.1

Type RM Length L Ch R = 1,297616,2510,2510,2510
BEGIN DESCRIPTION:
Clear Fork Brazos Rv 76.0
END DESCRIPTION:
XS GIS Cut Line= 2
      1649655.01      6997438.01      1647889.80      6996766.29
#Sta/Elev= 30
  4376.9 1507.80  4416.7 1494.46  4516.0 1473.68  4623.0 1471.06  4826.3 1472.12
  4866.4 1468.66  4879.8 1465.68  4896.0 1456.76  4951.3 1442.19  4960.0 1442.19
  4970.5 1441.19  5086.0 1442.19  5091.2 1446.25  5095.9 1446.03  5121.3 1456.86
  5126.6 1452.36  5136.6 1460.24  5146.0 1461.66  5151.4 1456.72  5158.0 1454.42
  5200.8 1457.24  5222.2 1469.55  5231.0 1470.73  5386.3 1471.15  5546.2 1477.17
  5576.3 1470.90  5631.1 1480.24  5703.7 1480.14  5935.6 1494.03  6265.6 1504.80
#Mann=6,-1,0
  4376.9    0.12       0  4896.0    0.05       0  4960.0    0.03       0
  5086.0    0.05       0  5095.9    0.12       0  5386.3    0.05       0
Bank Sta=4960,5086
Exp/Cntr=0.3,0.1

Type RM Length L Ch R = 1,295106,1666,1666,1666
BEGIN DESCRIPTION:
Mapping XS bf588705
END DESCRIPTION:
XS GIS Cut Line= 2
      1650798.72      6996683.46      1650332.18      6994632.86
#Sta/Elev= 30
  3621.6 1511.82  3986.1 1500.74  4204.2 1490.98  4333.4 1480.18  4338.5 1482.08
  4381.5 1473.49  4429.7 1468.35  4515.8 1465.41  4606.4 1467.53  4806.6 1472.52
  4827.1 1470.00  4857.9 1456.62  4888.6 1448.56  4930.1 1445.92  4968.1 1439.74
  4972.6 1438.74  5022.1 1439.74  5042.5 1452.89  5130.0 1476.09  5192.3 1486.92
  5240.5 1489.73  5319.4 1503.81  5360.4 1514.67  5460.9 1531.59  5509.1 1536.46
  5524.5 1542.69  5665.1 1580.25  5686.4 1591.25  5691.5 1590.74  5724.6 1608.33
#Mann=7,-1,0
  3621.6    0.05       0  4606.4    0.12       0  4930.1    0.05       0
  4968.1    0.05       0  5022.1    0.05       0  5130.0    0.12       0
  5665.1    0.05       0
Bank Sta=4968.1,5022.1
Exp/Cntr=0.3,0.1

Type RM Length L Ch R = 1,293440,2656,2656,2656
BEGIN DESCRIPTION:
Clear Fork Brazos Rv 75.0
END DESCRIPTION:
XS GIS Cut Line= 3
      1651454.99      6996388.01      1651955.00      6995888.00
      1651955.00      6995388.02
#Sta/Elev= 30
  4294.2 1487.09  4393.2 1480.37  4506.3 1475.25  4605.3 1469.53  4690.2 1465.95
  4748.1 1465.03  4817.5 1464.73  4902.3 1468.09  4916.5 1466.11  4930.6 1458.27
  4944.8 1453.30  4987.2 1450.48  4992.8 1439.56  5000.3 1438.56  5075.3 1438.56
  5082.8 1439.56  5111.3 1439.58  5121.3 1443.40  5131.3 1452.16  5161.3 1451.93
  5210.5 1458.19  5241.3 1464.79  5251.3 1468.13  5301.3 1480.44  5361.3 1500.76
  5411.3 1519.94  5461.3 1531.48  5488.9 1540.12  5498.8 1543.30  5501.3 1543.30
#Mann=6,-1,0
  4294.2    0.05       0  4748.1    0.12       0  4992.8    0.07       0
  5082.8    0.12       0  5210.5    0.12       0  5488.9    0.05       0
Bank Sta=4992.8,5082.8
Exp/Cntr=0.3,0.1

Type RM Length L Ch R = 1,290784,2703,2703,2703
BEGIN DESCRIPTION:
Mapping XS b72f16ef
END DESCRIPTION:
XS GIS Cut Line= 2
      1651319.54      6997692.61      1654260.03      6998658.30
#Sta/Elev= 30
  3311.6 1495.53  3527.9 1488.25  3612.1 1481.15  3821.5 1471.23  3928.6 1469.01
  4081.4 1466.82  4463.6 1466.92  4552.5 1465.09  4706.7 1463.26  4801.4 1452.07
  4816.7 1452.72  4832.1 1453.81  4864.6 1444.50  4875.1 1446.65  4913.6 1442.87
  4977.3 1442.36  4990.8 1438.63  4993.0 1437.63  5017.8 1438.63  5064.6 1448.48
  5085.6 1461.71  5104.5 1467.29  5275.1 1469.79  5475.1 1477.96  5643.5 1500.74
  5801.4 1526.70  6022.4 1551.06  6323.3 1594.13  6333.0 1595.20  6406.6 1615.87
#Mann=11,-1,0
  3311.6    0.05       0  3928.6    0.12       0  4081.4    0.05       0
  4463.6    0.12       0  4552.5    0.05       0  4816.7    0.12       0
  4832.1    0.05       0  4990.8    0.05       0  5017.8    0.05       0
  6323.3    0.12       0  6333.0    0.05       0
Bank Sta=4990.8,5017.8
Exp/Cntr=0.3,0.1

Type RM Length L Ch R = 1,288081,2331,2331,2331
BEGIN DESCRIPTION:
Mapping XS 7b2b0c0f
END DESCRIPTION:
XS GIS Cut Line= 2
      1651048.26      6999667.43      1653674.11      7000188.26
#Sta/Elev= 30
  4432.6 1526.44  4633.2 1517.78  4745.3 1506.78  4806.5 1488.84  4821.4 1486.08
  4847.3 1476.00  4872.6 1469.62  4877.8 1464.25  4949.2 1438.05  4969.6 1436.46
  4972.3 1434.67  4978.3 1433.67  5044.3 1434.67  5051.2 1434.67  5061.4 1439.15
  5071.5 1446.72  5080.0 1448.63  5102.1 1453.08  5128.5 1463.04  5216.5 1463.32
  5295.8 1459.38  5384.4 1465.50  5419.4 1465.24  5764.8 1463.97  5896.3 1464.86
  6080.8 1475.66  6692.5 1498.60  6827.9 1506.42  6896.4 1513.95  7109.6 1525.79
#Mann=7,-1,0
  4432.6    0.05       0  4972.3    0.05       0  5044.3    0.05       0
  5080.0    0.12       0  5216.5    0.05       0  5419.4    0.12       0
  5764.8    0.05       0
Bank Sta=4972.3,5044.3
Exp/Cntr=0.3,0.1

Type RM Length L Ch R = 1,285750,1536,1536,1536
BEGIN DESCRIPTION:
Clear Fork Brazos Rv 73.0
END DESCRIPTION:
XS GIS Cut Line= 3
      1651054.95      7002038.00      1651555.00      7002038.00
      1654554.97      7001538.00
#Sta/Elev= 30
  4499.1 1554.73  4599.1 1544.35  4649.1 1534.19  4849.1 1462.29  4919.1 1449.18
  4939.1 1437.06  4953.0 1434.39  4957.5 1433.39  5007.0 1434.39  5080.2 1439.21
  5093.9 1445.33  5100.5 1449.48  5130.9 1448.63  5171.5 1457.02  5330.2 1459.11
  5397.1 1462.63  5483.4 1460.90  5546.6 1460.66  5673.9 1468.79  5931.8 1479.80
  6431.1 1487.31  7067.3 1508.73  7343.5 1529.62  7460.1 1549.44  7513.4 1550.94
  7715.8 1585.03  7769.3 1594.98  7847.9 1620.32  7946.8 1634.75  8040.5 1638.15
#Mann=8,-1,0
  4499.1    0.05       0  4953.0    0.05       0  5007.0    0.05       0
  5093.9    0.12       0  5330.2    0.05       0  5483.4    0.12       0
  5673.9    0.05       0  7715.8    0.12       0
Bank Sta=4953,5007
Exp/Cntr=0.3,0.1

Type RM Length L Ch R = 1,284214,1531,1531,1531
BEGIN DESCRIPTION:
Mapping XS b1c2323f
END DESCRIPTION:
XS GIS Cut Line= 2
      1651211.99      7003628.76      1653601.32      7003005.86
#Sta/Elev= 30
  4029.2 1567.82  4049.9 1566.26  4055.1 1568.71  4090.4 1562.78  4095.6 1563.77
  4247.2 1525.95  4352.7 1504.00  4485.0 1468.99  4525.4 1463.68  4654.8 1462.03
  4687.4 1462.31  4745.4 1450.88  4776.4 1448.18  4878.5 1445.72  4910.7 1445.48
  4959.5 1432.31  4965.5 1431.31  5031.5 1432.31  5032.4 1432.43  5046.6 1436.14
  5055.4 1445.16  5082.0 1449.36  5087.1 1454.10  5096.7 1457.17  5122.4 1460.01
  5196.5 1461.19  5427.4 1466.71  5916.7 1490.05  6351.8 1500.81  6498.4 1507.85
#Mann=7,-1,0
  4029.2    0.05       0  4654.8    0.12       0  4878.5    0.05       0
  4959.5    0.05       0  5031.5    0.05       0  5032.4    0.12       0
  5196.5    0.05       0
Bank Sta=4959.5,5031.5
Exp/Cntr=0.3,0.1

Type RM Length L Ch R = 1,282683,2028,2028,2028
BEGIN DESCRIPTION:
Mapping XS b9bf7f8e
END DESCRIPTION:
XS GIS Cut Line= 2
      1651059.14      7004799.82      1653478.84      7004669.61
#Sta/Elev= 30
  3455.5 1590.94  3681.7 1538.68  3872.0 1505.34  3992.1 1471.07  4062.2 1458.74
  4102.3 1448.73  4132.3 1448.81  4262.5 1460.76  4352.7 1462.87  4452.8 1450.41
  4723.2 1442.84  4763.3 1436.48  4783.3 1439.86  4825.0 1440.64  4903.5 1438.47
  4924.3 1434.44  4995.6 1431.52  5000.8 1430.52  5058.6 1431.52  5063.7 1435.88
  5069.9 1448.34  5074.9 1443.49  5083.7 1461.86  5269.0 1458.74  5475.2 1461.24
  5554.4 1464.32  5654.5 1484.81  5704.6 1486.02  5764.7 1483.19  5878.7 1487.23
#Mann=7,-1,0
  3455.5    0.05       0  4825.0    0.12       0  4924.3    0.05       0
  4995.6    0.05       0  5058.6    0.05       0  5269.0    0.12       0
  5475.2    0.05       0
Bank Sta=4995.6,5058.6
Exp/Cntr=0.3,0.1

Type RM Length L Ch R = 1,280655,2811,2811,2811
BEGIN DESCRIPTION:
Mapping XS ae6b22d2
END DESCRIPTION:
XS GIS Cut Line= 3
      1650960.89      7006540.22      1651916.35      7006557.63
      1654444.52      7005971.70
#Sta/Elev= 30
  2774.0 1507.96  2938.1 1498.99  3118.2 1477.27  3488.2 1470.65  4327.3 1465.30
  4570.0 1458.80  4600.8 1451.19  4611.0 1454.36  4641.8 1442.51  4672.6 1440.80
  4693.1 1431.01  4734.2 1434.57  4754.7 1442.79  4913.2 1437.73  4970.3 1435.56
  4980.6 1434.15  4980.9 1429.37  4985.4 1428.37  5034.9 1429.37  5078.5 1445.54
  5185.4 1446.29  5259.4 1449.81  5288.5 1444.38  5360.4 1450.34  5422.0 1478.56
  5452.8 1485.77  5729.9 1492.85  5935.2 1505.02  6078.9 1518.17  6324.8 1531.85
#Mann=6,-1,0
  2774.0    0.05       0  4754.7    0.12       0  4913.2    0.05       0
  4980.9    0.07       0  5034.9    0.05       0  5185.4    0.05       0
Bank Sta=4980.9,5034.9
Exp/Cntr=0.3,0.1

Type RM Length L Ch R = 1,277844,3247,3247,3247
BEGIN DESCRIPTION:
Mapping XS 60efb378
END DESCRIPTION:
XS GIS Cut Line= 2
      1651872.96      7008651.81      1655051.12      7008250.47
#Sta/Elev= 30
  4329.5 1604.13  4351.7 1602.35  4492.8 1537.26  4639.1 1489.89  4734.7 1465.08
  4879.8 1446.69  4906.1 1433.82  4926.2 1428.05  4944.0 1427.93  4960.8 1424.61
  4964.6 1423.61  5005.8 1424.61  5017.0 1433.79  5027.0 1437.49  5057.3 1438.60
  5067.4 1434.41  5079.7 1436.88  5127.8 1440.83  5179.9 1439.08  5200.7 1437.19
  5280.1 1441.13  5319.3 1445.95  5480.6 1451.56  5531.0 1457.48  5964.4 1477.59
  6297.0 1486.86  6901.8 1491.43  7196.3 1503.36  7431.9 1521.23  7532.9 1525.61
#Mann=7,-1,0
  4329.5    0.05       0  4944.0    0.12       0  4960.8    0.07       0
  5005.8    0.12       0  5079.7    0.05       0  5179.9    0.12       0
  5280.1    0.05       0
Bank Sta=4960.8,5005.8
Exp/Cntr=0.3,0.1

Type RM Length L Ch R = 1,274597,2415,2415,2415
BEGIN DESCRIPTION:
Mapping XS a070693c
END DESCRIPTION:
XS GIS Cut Line= 3
      1653836.92      7011917.87      1654835.18      7010507.28
      1655703.23      7009758.59
#Sta/Elev= 30
  3888.9 1568.05  3945.0 1563.02  4123.4 1523.68  4381.9 1481.31  4806.6 1456.18
  4905.6 1437.01  4934.5 1438.53  4965.2 1424.39  4972.7 1423.39  5055.2 1424.39
  5071.2 1441.40  5092.5 1443.01  5158.5 1452.55  5236.3 1452.65  5279.2 1445.99
  5293.9 1435.40  5300.1 1439.25  5308.7 1432.87  5314.8 1437.17  5329.6 1432.47
  5350.5 1434.92  5371.4 1442.88  5380.1 1450.82  5466.2 1455.22  6190.6 1459.85
  6254.3 1465.20  6346.4 1483.91  6432.0 1495.42  6594.3 1508.04  6763.3 1511.72
#Mann=5,-1,0
  3888.9    0.05       0  4965.2    0.05       0  5055.2    0.05       0
  5092.5    0.12       0  5158.5    0.05       0
Bank Sta=4965.2,5055.2
Exp/Cntr=0.3,0.1

Type RM Length L Ch R = 1,272182,1850,1850,1850
BEGIN DESCRIPTION:
Mapping XS 6e7a28cb
END DESCRIPTION:
XS GIS Cut Line= 3
      1654439.71      7012800.34      1655537.36      7012884.06
      1657490.34      7011033.38
#Sta/Elev= 30
  2366.8 1508.65  2462.4 1505.39  2652.9 1489.06  2943.8 1477.84  3505.7 1474.36
  3901.8 1458.35  4283.7 1452.33  4828.3 1451.76  4878.6 1446.84  4912.1 1439.18
  4927.3 1437.93  4941.5 1428.41  4991.2 1428.05  4993.7 1424.33  4997.4 1423.33
  5038.7 1424.33  5062.0 1429.03  5076.1 1427.94  5155.3 1451.72  5203.2 1472.47
  5231.5 1479.21  5309.6 1514.82  5385.5 1523.05  5571.3 1537.95  5606.5 1545.90
  5719.7 1559.28  5833.0 1580.82  5868.2 1591.73  5945.9 1602.04  6158.2 1615.77
#Mann=7,-1,0
  2366.8    0.05       0  4878.6    0.12       0  4912.1    0.05       0
  4993.7    0.05       0  5038.7    0.05       0  5155.3    0.12       0
  5385.5    0.05       0
Bank Sta=4993.7,5038.7
Exp/Cntr=0.3,0.1

Type RM Length L Ch R = 1,270332,3838,3838,3838
BEGIN DESCRIPTION:
Clear Fork Brazos Rv 69.0
END DESCRIPTION:
XS GIS Cut Line= 3
      1654496.48      7013014.51      1657455.00      7013138.00
      1657955.01      7013138.00
#Sta/Elev= 30
  2037.0 1505.61  2075.5 1504.94  2240.6 1494.95  2345.8 1484.42  2556.0 1477.10
  2856.2 1473.91  3200.6 1474.79  3486.8 1459.62  3606.9 1455.57  4007.2 1454.88
  4227.4 1451.79  4407.6 1452.46  4635.6 1448.87  4787.9 1451.00  4817.9 1446.75
  4886.7 1443.94  4908.0 1442.71  4948.0 1424.15  4954.5 1422.59  4960.5 1421.59
  5026.5 1422.59  5038.1 1427.02  5103.2 1429.03  5118.1 1430.12  5138.1 1436.78
  5165.7 1439.00  5208.1 1443.41  5248.1 1454.10  5358.1 1509.13  5498.1 1515.25
#Mann=6,-1,0
  2037.0    0.05       0  4886.7    0.12       0  4954.5    0.05       0
  5026.5    0.12       0  5103.2    0.12       0  5165.7    0.05       0
Bank Sta=4954.5,5026.5
Exp/Cntr=0.3,0.1

Type RM Length L Ch R = 1,266494,3051,3051,3051
BEGIN DESCRIPTION:
Clear Fork Brazos Rv 68.0
END DESCRIPTION:
XS GIS Cut Line= 3
      1654754.97      7015687.98      1656755.00      7016688.00
      1657255.00      7016688.00
#Sta/Elev= 30
  2749.4 1504.56  2869.6 1497.00  2942.3 1494.15  3003.8 1487.14  3062.5 1483.12
  3465.0 1467.19  3702.6 1454.74  3724.9 1455.56  3741.7 1453.12  3769.6 1452.02
  4127.4 1445.94  4597.0 1447.44  4747.9 1449.39  4887.7 1447.59  4940.8 1436.83
  4954.8 1426.18  4961.7 1418.17  4967.7 1417.17  5033.7 1418.17  5055.5 1419.67
  5065.5 1423.22  5116.6 1432.51  5145.5 1433.86  5185.5 1438.72  5235.5 1448.23
  5285.5 1467.02  5325.5 1486.10  5375.5 1503.87  5435.5 1523.21  5485.5 1532.47
#Mann=5,-1,0
  2749.4    0.05       0  4887.7    0.12       0  4961.7    0.07       0
  5033.7    0.12       0  5116.6    0.05       0
Bank Sta=4961.7,5033.7
Exp/Cntr=0.3,0.1

Type RM Length L Ch R = 1,263443,2042,2042,2042
BEGIN DESCRIPTION:
Clear Fork Brazos Rv 67.0
END DESCRIPTION:
XS GIS Cut Line= 3
      1654455.04      7018888.00      1655508.43      7018915.31
      1657955.02      7019888.01
#Sta/Elev= 30
  4249.3 1482.37  4499.3 1468.04  4559.4 1469.15  4647.4 1455.33  4799.4 1424.84
  4819.5 1427.11  4856.9 1422.07  4969.5 1422.43  4982.8 1417.57  4984.9 1416.79
  4987.1 1415.79  5011.9 1416.79  5019.5 1419.30  5029.5 1430.48  5039.5 1432.51
  5089.5 1435.89  5139.6 1447.46  5194.7 1446.80  5697.5 1442.71  6355.9 1448.95
  6488.1 1455.93  6566.4 1473.30  6620.4 1481.60  6655.4 1480.74  6704.0 1492.61
  7081.8 1502.05  7297.7 1503.98  7548.6 1494.50  7774.5 1498.78  7935.9 1494.07
#Mann=7,-1,0
  4249.3    0.05       0  4647.4    0.12       0  4856.9    0.05       0
  4982.8    0.12       0  4984.9    0.07       0  5011.9    0.12       0
  5194.7    0.05       0
Bank Sta=4984.9,5011.9
Exp/Cntr=0.3,0.1

Type RM Length L Ch R = 1,261401,2642,2642,2642
BEGIN DESCRIPTION:
Mapping XS f546d4a1
END DESCRIPTION:
XS GIS Cut Line= 3
      1654607.32      7020815.44      1655431.97      7020142.70
      1657361.74      7019958.39
#Sta/Elev= 30
  4236.0 1570.31  4317.9 1574.28  4396.2 1570.05  4559.2 1545.76  4680.5 1497.68
  4730.1 1470.28  4814.8 1438.99  4829.1 1434.21  4936.1 1419.50  4949.9 1413.95
  4954.4 1412.95  5003.9 1413.95  5020.9 1415.36  5043.1 1430.86  5062.5 1434.01
  5082.2 1439.47  5092.7 1442.78  5241.3 1445.26  5494.2 1441.03  5544.4 1447.00
  5624.8 1431.87  5664.9 1433.93  5705.1 1446.04  5755.3 1440.66  5976.3 1446.35
  6408.3 1445.07  6518.8 1450.53  6669.5 1470.77  6772.3 1477.11  7238.8 1492.42
#Mann=5,-1,0
  4236.0    0.05       0  4949.9    0.05       0  5003.9    0.05       0
  5062.5    0.12       0  5082.2    0.05       0
Bank Sta=4949.9,5003.9
Exp/Cntr=0.3,0.1

Type RM Length L Ch R = 1,258759,2942,2942,2942
BEGIN DESCRIPTION:
Clear Fork Brazos Rv 66.0
END DESCRIPTION:
XS GIS Cut Line= 3
      1657004.98      7021988.03      1657505.00      7020988.00
      1657505.00      7020487.97
#Sta/Elev= 30
  3882.3 1576.88  4008.1 1572.87  4142.3 1572.28  4270.9 1532.69  4388.2 1503.49
  4405.0 1495.66  4433.0 1487.74  4472.1 1472.18  4477.7 1471.96  4494.5 1461.84
  4500.1 1461.80  4539.2 1444.50  4544.8 1444.41  4561.5 1437.09  4583.9 1432.79
  4628.6 1429.68  4813.1 1427.97  4897.0 1421.81  4947.3 1420.58  4975.8 1412.92
  4981.0 1411.92  5038.8 1412.92  5090.4 1432.32  5140.4 1441.52  5182.2 1444.18
  5320.4 1451.06  5380.4 1451.58  5441.7 1458.15  5454.2 1459.40  5500.4 1464.88
#Mann=6,-1,0
  3882.3    0.05       0  4975.8    0.07       0  5038.8    0.05       0
  5182.2    0.05       0  5441.7    0.12       0  5454.2    0.05       0
Bank Sta=4975.8,5038.8
Exp/Cntr=0.3,0.1

Type RM Length L Ch R = 1,255817,1831,1831,1831
BEGIN DESCRIPTION:
Mapping XS cb9af0e1
END DESCRIPTION:
XS GIS Cut Line= 2
      1660495.61      7021744.58      1659599.31      7019775.26
#Sta/Elev= 30
  3677.2 1480.09  3683.6 1480.70  3805.3 1471.26  3857.2 1455.33  3960.4 1444.99
  3978.0 1447.87  4121.8 1440.69  4564.3 1438.33  4731.2 1434.05  4748.8 1427.10
  4777.4 1425.73  4800.4 1431.80  4915.0 1434.21  4958.9 1425.12  4972.8 1411.81
  4980.9 1413.54  4985.9 1409.56  4988.9 1408.56  5021.9 1409.56  5070.5 1416.14
  5093.6 1411.58  5111.1 1414.17  5139.7 1411.43  5168.2 1420.02  5200.6 1417.22
  5222.6 1426.13  5237.4 1426.05  5404.3 1464.87  5674.4 1464.31  5840.9 1475.90
#Mann=4,-1,0
  3677.2    0.12       0  3683.6    0.05       0  4985.9    0.05       0
  5021.9    0.05       0
Bank Sta=4985.9,5021.9
Exp/Cntr=0.3,0.1

Type RM Length L Ch R = 1,253986,2141,2141,2141
BEGIN DESCRIPTION:
Clear Fork Brazos Rv 65.0
END DESCRIPTION:
XS GIS Cut Line= 2
      1661254.99      7021788.04      1661845.17      7019367.45
#Sta/Elev= 30
  3755.9 1510.32  3879.5 1487.24  3987.8 1461.82  4071.2 1448.95  4706.9 1434.63
  4743.5 1426.25  4754.4 1419.98  4774.9 1419.62  4795.5 1429.88  4816.1 1433.49
  4888.2 1437.40  4898.5 1436.81  4920.5 1426.66  4962.2 1419.72  4983.1 1406.35
  4986.8 1405.35  5028.1 1406.35  5063.1 1409.84  5073.4 1416.51  5123.9 1429.42
  5149.6 1431.42  5152.8 1431.63  5295.8 1441.16  5379.2 1440.09  5551.1 1448.53
  5931.5 1474.09  6014.9 1484.47  6071.8 1499.73  6145.1 1508.21  6247.4 1530.54
#Mann=5,-1,0
  3755.9    0.05       0  4983.1    0.05       0  5028.1    0.05       0
  5149.6    0.12       0  5152.8    0.05       0
Bank Sta=4983.1,5028.1
Exp/Cntr=0.3,0.1

Type RM Length L Ch R = 1,251845,1477,1477,1477
BEGIN DESCRIPTION:
Mapping XS 1c7c4698
END DESCRIPTION:
XS GIS Cut Line= 2
      1663743.62      7021325.45      1662669.85      7019503.30
#Sta/Elev= 30
  4395.8 1465.78  4545.2 1463.25  4625.2 1459.03  4822.3 1444.71  4832.2 1443.64
  4847.6 1438.99  4880.9 1424.74  4912.2 1421.07  4939.5 1413.52  4955.1 1412.57
  4970.0 1406.27  4975.3 1405.27  5033.0 1406.27  5056.6 1420.93  5087.9 1424.67
  5093.7 1427.32  5113.4 1431.33  5146.5 1433.56  5228.8 1433.84  5562.2 1438.31
  5897.9 1449.05  6226.8 1455.58  6276.6 1459.50  6319.6 1466.06  6356.6 1468.14
  6372.2 1471.89  6415.2 1475.36  6467.9 1485.53  6473.7 1485.01  6510.8 1490.36
#Mann=6,-1,0
  4395.8    0.05       0  4847.6    0.12       0  4970.0    0.05       0
  5033.0    0.12       0  5113.4    0.12       0  5228.8    0.05       0
Bank Sta=4970,5033
Exp/Cntr=0.3,0.1

Type RM Length L Ch R = 1,250368,1000,1000,1000
BEGIN DESCRIPTION:
Mapping XS 7949a791
END DESCRIPTION:
XS GIS Cut Line= 3
      1663946.20      7021274.31      1664234.56      7020706.89
      1664346.13      7019572.56
#Sta/Elev= 30
  3438.1 1465.11  3904.8 1461.93  4123.7 1456.91  4314.6 1450.28  4364.9 1447.39
  4433.4 1439.37  4495.5 1436.29  4505.6 1434.56  4534.7 1433.15  4539.8 1435.03
  4555.8 1434.68  4565.8 1433.61  4575.9 1429.74  4636.1 1425.44  4736.7 1421.37
  4843.7 1421.23  4897.4 1419.51  4937.6 1413.35  4977.8 1409.98  4987.9 1407.56
  4994.9 1403.87  4997.2 1402.87  5021.9 1403.87  5038.1 1404.69  5074.5 1412.34
  5098.4 1424.03  5128.5 1430.57  5152.7 1433.99  5188.8 1449.28  5214.4 1457.47
#Mann=4,-1,0
  3438.1    0.05       0  4994.9    0.05       0  5021.9    0.05       0
  5074.5    0.12       0
Bank Sta=4994.9,5021.9
Exp/Cntr=0.3,0.1

Type RM Length L Ch R = 1,249368,2205,2205,2205
BEGIN DESCRIPTION:
Mapping XS 457d8ec2
END DESCRIPTION:
XS GIS Cut Line= 2
      1664221.05      7021010.74      1665436.31      7020055.90
#Sta/Elev= 30
  3995.3 1462.14  4334.4 1456.79  4676.1 1441.10  4791.9 1429.48  4798.0 1430.94
  4804.4 1427.17  4862.2 1418.45  4904.9 1417.76  4918.3 1415.89  4926.4 1418.54
  4940.8 1414.88  4954.1 1403.43  4970.8 1402.13  4974.6 1401.13  5015.8 1402.13
  5017.7 1406.66  5061.1 1410.43  5081.9 1417.48  5146.0 1421.86  5183.0 1437.21
  5210.2 1442.29  5259.9 1461.13  5296.9 1466.20  5317.7 1474.15  5367.4 1485.89
  5402.7 1498.93  5424.7 1502.08  5481.3 1526.60  5536.8 1559.15  5540.8 1559.15
#Mann=5,-1,0
  3995.3    0.05       0  4791.9    0.12       0  4904.9    0.05       0
  4970.8    0.05       0  5015.8    0.12       0
Bank Sta=4970.8,5015.8
Exp/Cntr=0.3,0.1

Type RM Length L Ch R = 1,247163,2158,2158,2158
BEGIN DESCRIPTION:
Clear Fork Brazos Rv 64.0
END DESCRIPTION:
XS GIS Cut Line= 4
      1664262.67      7022438.00      1664955.00      7022438.00
      1665455.00      7022438.00      1665954.97      7022438.00
#Sta/Elev= 30
  3807.5 1474.54  3929.8 1472.13  4009.8 1465.51  4129.8 1461.05  4149.8 1458.18
  4209.8 1442.45  4239.8 1439.87  4349.8 1437.51  4559.8 1439.82  4909.8 1432.44
  4929.8 1430.28  4959.8 1419.17  4979.8 1400.37  4984.8 1401.16  4992.3 1399.16
  5067.3 1399.16  5074.8 1401.16  5079.8 1409.52  5089.8 1412.54  5109.8 1410.15
  5119.8 1412.33  5169.8 1431.10  5199.8 1444.06  5209.8 1451.43  5229.8 1458.99
  5298.2 1473.73  5339.8 1484.04  5399.8 1495.34  5469.8 1513.51  5499.8 1519.32
#Mann=4,-1,0
  3807.5    0.05       0  4984.8    0.03       0  5074.8    0.05       0
  5298.2    0.05       0
Bank Sta=4984.8,5074.8
Exp/Cntr=0.3,0.1

Type RM Length L Ch R = 1,245005,2135,2135,2135
BEGIN DESCRIPTION:
Mapping XS 14316226
END DESCRIPTION:
XS GIS Cut Line= 2
      1664307.87      7023983.87      1665403.72      7024830.17
#Sta/Elev= 30
  4247.0 1452.46  4397.1 1446.56  4483.4 1445.12  4520.5 1441.88  4569.2 1436.35
  4683.3 1431.18  4753.9 1429.79  4882.5 1430.66  4888.9 1426.47  4903.4 1421.05
  4938.7 1418.88  4967.7 1406.77  4975.8 1400.03  4978.0 1400.03  4985.5 1399.03
  5068.0 1400.03  5089.9 1414.82  5110.8 1413.40  5146.1 1418.71  5160.6 1412.62
  5166.9 1413.38  5239.4 1443.48  5307.3 1453.14  5353.5 1462.16  5409.6 1468.04
  5438.6 1473.35  5459.5 1474.21  5488.4 1479.52  5602.6 1492.69  5631.6 1494.43
#Mann=5,-1,0
  4247.0    0.05       0  4520.5    0.12       0  4978.0    0.07       0
  5068.0    0.12       0  5307.3    0.05       0
Bank Sta=4978,5068
Exp/Cntr=0.3,0.1

Type RM Length L Ch R = 1,242870,466,466,466
BEGIN DESCRIPTION:
Mapping XS 5613bd06
END DESCRIPTION:
XS GIS Cut Line= 3
      1663222.18      7025168.64      1663472.34      7025589.75
      1664122.60      7026684.36
#Sta/Elev= 30
  3867.6 1445.86  4006.4 1443.63  4037.5 1440.17  4111.1 1441.15  4157.2 1439.03
  4292.7 1438.62  4473.9 1442.09  4563.6 1440.36  4670.7 1433.24  4774.1 1429.91
  4867.4 1417.03  4921.0 1416.56  4948.6 1416.76  4971.8 1407.91  4978.5 1400.57
  4992.8 1399.93  4999.6 1398.93  5073.8 1399.93  5079.8 1399.93  5088.2 1404.39
  5095.4 1412.71  5103.5 1417.47  5116.8 1423.23  5132.4 1425.57  5181.2 1426.64
  5196.7 1431.19  5233.7 1449.58  5273.8 1457.46  5402.2 1464.52  5630.6 1471.28
#Mann=7,-1,0
  3867.6    0.05       0  4157.2    0.12       0  4921.0    0.05       0
  4992.8    0.03       0  5073.8    0.05       0  5103.5    0.12       0
  5273.8    0.05       0
Bank Sta=4992.8,5073.8
Exp/Cntr=0.3,0.1

Type RM Length L Ch R = 1,242404,1489,1489,1489
BEGIN DESCRIPTION:
Mapping XS 25fb7d25
END DESCRIPTION:
XS GIS Cut Line= 3
      1662558.00      7024665.42      1662857.89      7026018.23
      1664002.05      7026864.72
#Sta/Elev= 30
  2851.3 1471.00  2903.4 1463.97  3017.8 1456.54  3321.3 1444.91  3560.7 1439.82
  4093.4 1438.03  4123.2 1437.90  4242.3 1435.58  4335.3 1425.04  4357.1 1421.35
  4363.3 1416.72  4392.6 1416.46  4444.7 1425.37  4489.6 1428.08  4835.1 1429.19
  4855.9 1426.09  4864.3 1421.86  4870.5 1423.40  4878.9 1418.65  4914.4 1413.96
  4927.4 1399.91  4935.7 1398.91  5026.4 1399.91  5048.4 1412.32  5121.0 1421.27
  5164.9 1433.16  5188.8 1443.77  5221.2 1450.94  5292.2 1455.46  5660.2 1467.50
#Mann=10,-1,0
  2851.3    0.05       0  4093.4    0.12       0  4123.2    0.05       0
  4335.3    0.12       0  4444.7    0.05       0  4489.6    0.12       0
  4927.4    0.03       0  5026.4    0.12       0  5048.4    0.12       0
  5188.8    0.05       0
Bank Sta=4927.4,5026.4
Exp/Cntr=0.3,0.1

Type RM Length L Ch R = 1,240915,1512,1512,1512
BEGIN DESCRIPTION:
Mapping XS af8a4a53
END DESCRIPTION:
XS GIS Cut Line= 2
      1661855.58      7027282.46      1663450.27      7027434.33
#Sta/Elev= 30
  4495.4 1526.96  4497.6 1526.96  4500.5 1522.06  4505.5 1522.94  4555.1 1505.24
  4575.2 1502.17  4603.5 1494.67  4608.5 1495.41  4711.4 1466.91  4725.9 1466.29
  4776.1 1455.75  4819.4 1444.67  4826.3 1440.68  4876.5 1428.63  4896.6 1420.74
  4956.9 1414.51  4977.0 1407.93  4987.7 1397.56  4991.5 1396.56  5032.7 1397.56
  5047.3 1399.63  5097.5 1401.42  5133.3 1407.33  5138.4 1406.45  5187.9 1410.99
  5452.3 1420.57  5640.0 1429.34  5891.1 1446.66  5977.1 1448.84  6097.3 1449.01
#Mann=3,-1,0
  4495.4    0.05       0  4987.7    0.05       0  5032.7    0.05       0
Bank Sta=4987.7,5032.7
Exp/Cntr=0.3,0.1

Type RM Length L Ch R = 1,239403,2127,2127,2127
BEGIN DESCRIPTION:
Clear Fork Brazos Rv 62.0
END DESCRIPTION:
XS GIS Cut Line= 3
      1662805.03      7028937.97      1663305.00      7028438.00
      1663805.02      7027937.98
#Sta/Elev= 30
  4287.4 1591.81  4343.9 1580.08  4400.5 1573.42  4457.1 1563.71  4499.5 1559.08
  4570.2 1555.29  4640.9 1542.86  4697.5 1522.32  4782.3 1480.52  4867.2 1446.76
  4909.6 1419.46  4966.2 1400.55  4990.9 1398.50  4992.8 1395.79  4995.8 1394.79
  5028.8 1395.79  5079.3 1402.84  5107.6 1399.54  5135.9 1412.64  5164.2 1413.08
  5192.5 1423.68  5206.6 1425.20  5220.7 1420.65  5234.9 1424.28  5263.2 1427.14
  5412.7 1432.69  5432.9 1431.78  5572.0 1437.37  5656.3 1441.92  5701.6 1444.16
#Mann=6,-1,0
  4287.4    0.05       0  4992.8    0.07       0  5028.8    0.05       0
  5412.7    0.05       0  5572.0    0.12       0  5656.3    0.05       0
Bank Sta=4992.8,5028.8
Exp/Cntr=0.3,0.1

Type RM Length L Ch R = 1,237276,1747,1747,1747
BEGIN DESCRIPTION:
Mapping XS b8ccc999
END DESCRIPTION:
XS GIS Cut Line= 2
      1665262.70      7029409.20      1665295.24      7028042.48
#Sta/Elev= 30
  4479.8 1560.24  4501.0 1555.63  4521.0 1548.58  4561.0 1532.66  4631.0 1509.03
  4671.1 1491.40  4716.6 1476.14  4771.1 1463.22  4786.3 1456.94  4791.3 1458.40
  4814.5 1451.20  4831.1 1443.04  4841.1 1434.59  4891.1 1410.87  4912.3 1406.65
  4949.7 1392.24  4954.2 1391.24  5003.7 1392.24  5010.1 1396.55  5021.2 1396.71
  5031.2 1401.81  5041.2 1404.11  5051.2 1410.06  5091.2 1422.96  5120.3 1423.51
  5281.2 1426.25  5551.3 1432.96  5694.7 1439.70  5758.9 1444.11  5846.9 1450.56
#Mann=11,-1,0
  4479.8    0.05       0  4716.6    0.12       0  4814.5    0.05       0
  4912.3    0.12       0  4949.7    0.07       0  5003.7    0.12       0
  5010.1     0.1       0  5120.3    0.12       0  5281.2    0.05       0
  5694.7    0.12       0  5758.9    0.05       0
Bank Sta=4949.7,5003.7
Exp/Cntr=0.3,0.1

Type RM Length L Ch R = 1,235529,2060,2060,2060
BEGIN DESCRIPTION:
Clear Fork Brazos Rv 61.0
END DESCRIPTION:
XS GIS Cut Line= 3
      1667254.97      7028637.97      1666755.00      7028138.00
      1666353.54      7027712.16
#Sta/Elev= 30
  4293.3 1530.00  4392.2 1513.79  4448.8 1497.45  4463.0 1490.89  4491.2 1481.98
  4547.8 1471.74  4604.4 1458.69  4689.2 1424.36  4717.5 1419.21  4774.1 1415.71
  4787.1 1416.83  4858.9 1414.05  4887.2 1410.34  4943.8 1408.74  4957.9 1406.71
  4972.1 1401.99  4991.3 1391.30  4997.3 1390.30  5063.3 1391.30  5071.0 1393.01
  5092.4 1404.19  5099.3 1403.90  5106.6 1408.52  5113.4 1406.62  5120.7 1408.59
  5155.9 1410.11  5205.7 1423.15  5240.9 1428.89  5522.3 1447.70  5585.6 1451.73
#Mann=5,-1,0
  4293.3    0.05       0  4787.1    0.12       0  4991.3    0.07       0
  5063.3    0.05       0  5522.3    0.05       0
Bank Sta=4991.3,5063.3
Exp/Cntr=0.3,0.1

Type RM Length L Ch R = 1,233469,1770,1770,1770
BEGIN DESCRIPTION:
Mapping XS bb9c758b
END DESCRIPTION:
XS GIS Cut Line= 2
      1668713.25      7027206.52      1667324.72      7026262.75
#Sta/Elev= 30
  4335.3 1514.15  4454.2 1504.82  4484.1 1500.56  4499.0 1495.22  4535.0 1488.32
  4612.9 1477.96  4678.7 1473.41  4720.6 1459.77  4750.5 1443.24  4772.8 1435.77
  4801.4 1423.13  4873.2 1410.28  4888.2 1404.47  4894.2 1404.32  4909.2 1412.16
  4951.1 1407.00  4966.1 1401.54  4979.2 1390.67  4983.7 1389.67  5033.2 1390.67
  5046.6 1392.80  5052.9 1398.65  5125.5 1405.47  5217.6 1409.27  5269.5 1415.44
  5304.4 1416.68  5325.3 1423.84  5348.8 1427.28  5418.0 1430.14  6014.2 1455.38
#Mann=7,-1,0
  4335.3    0.05       0  4772.8    0.12       0  4979.2    0.07       0
  5033.2    0.12       0  5125.5    0.05       0  5269.5    0.12       0
  5418.0    0.05       0
Bank Sta=4979.2,5033.2
Exp/Cntr=0.3,0.1

Type RM Length L Ch R = 1,231699,1982,1982,1982
BEGIN DESCRIPTION:
Clear Fork Brazos Rv 60.0
END DESCRIPTION:
XS GIS Cut Line= 4
      1669304.98      7025238.00      1668805.00      7025238.00
      1668305.00      7025238.00      1667434.88      7025238.00
#Sta/Elev= 30
  4493.4 1489.72  4573.4 1482.47  4613.4 1473.96  4653.4 1470.59  4693.4 1457.71
  4786.5 1437.28  4873.4 1423.44  4906.0 1414.76  4923.4 1406.91  4943.4 1402.80
  4963.4 1391.29  4968.4 1390.55  4975.9 1389.55  5058.4 1390.55  5063.4 1396.04
  5076.3 1404.18  5083.4 1406.15  5108.3 1407.41  5123.4 1410.48  5153.4 1420.21
  5173.4 1423.20  5248.9 1423.00  5256.5 1422.99  5403.4 1422.00  5763.4 1431.60
  5793.4 1434.88  5863.4 1448.12  5913.4 1453.54  6313.4 1483.57  6363.5 1483.92
#Mann=9,-1,0
  4493.4    0.05       0  4786.5    0.12       0  4906.0    0.05       0
  4968.4    0.03       0  5058.4    0.05       0  5076.3    0.12       0
  5108.3    0.05       0  5248.9    0.12       0  5256.5    0.05       0
Bank Sta=4968.4,5058.4
Exp/Cntr=0.3,0.1

Type RM Length L Ch R = 1,229717,1851,1851,1851
BEGIN DESCRIPTION:
Mapping XS 8812f60a
END DESCRIPTION:
XS GIS Cut Line= 2
      1669885.07      7023549.81      1667998.54      7023430.55
#Sta/Elev= 30
  3667.4 1484.99  3727.6 1483.49  3774.0 1475.49  3797.7 1473.72  3807.7 1472.11
  3837.8 1461.34  3877.9 1453.65  3918.0 1442.49  3988.1 1432.49  4028.2 1429.48
  4479.1 1415.05  4669.5 1419.26  4771.5 1419.24  4849.8 1419.73  4884.9 1418.02
  4899.9 1408.75  4928.0 1399.90  4940.0 1397.59  4950.5 1388.68  4957.3 1387.68
  5031.5 1388.68  5044.3 1393.33  5050.2 1402.60  5060.2 1407.35  5160.4 1440.91
  5210.5 1455.88  5250.6 1460.12  5330.8 1462.71  5431.0 1469.78  5557.7 1476.14
#Mann=5,-1,0
  3667.4    0.05       0  4771.5    0.12       0  4928.0    0.05       0
  4950.5    0.03       0  5031.5    0.05       0
Bank Sta=4950.5,5031.5
Exp/Cntr=0.3,0.1

Type RM Length L Ch R = 1,227866,2011,2011,2011
BEGIN DESCRIPTION:
Mapping XS fc679ce0
END DESCRIPTION:
XS GIS Cut Line= 2
      1670047.88      7022030.73      1668008.97      7021477.62
#Sta/Elev= 30
  3990.1 1497.11  4024.5 1495.78  4053.9 1488.16  4059.1 1489.08  4093.8 1477.75
  4098.9 1478.89  4138.8 1468.63  4158.9 1460.33  4247.9 1443.10  4402.0 1429.68
  4441.8 1423.31  4476.4 1414.11  4521.5 1411.98  4665.2 1420.33  4819.3 1413.66
  4864.3 1413.97  4925.6 1401.97  4938.7 1397.72  4946.3 1390.17  4963.5 1387.59
  4971.0 1386.59  5053.5 1387.59  5060.3 1398.37  5070.7 1404.15  5101.8 1416.24
  5112.1 1417.90  5174.3 1420.24  5475.5 1421.90  5733.5 1456.36  6102.7 1472.70
#Mann=3,-1,0
  3990.1    0.05       0  4963.5    0.03       0  5053.5    0.05       0
Bank Sta=4963.5,5053.5
Exp/Cntr=0.3,0.1

Type RM Length L Ch R = 1,225855,1886,1886,1886
BEGIN DESCRIPTION:
Mapping XS 28527f64
END DESCRIPTION:
XS GIS Cut Line= 2
      1670264.90      7020424.82      1668040.47      7019828.02
#Sta/Elev= 30
  3901.4 1479.56  3987.5 1474.45  4191.2 1438.67  4409.3 1425.20  4554.9 1419.58
  4761.6 1414.47  4858.9 1416.44  4916.5 1416.02  4926.3 1412.92  4946.1 1399.28
  4951.3 1399.31  4967.7 1389.32  4982.9 1386.49  4988.2 1385.49  5045.9 1386.49
  5050.6 1386.49  5066.1 1393.92  5092.0 1396.36  5100.9 1400.30  5172.5 1402.07
  5261.0 1400.78  5335.8 1403.59  5375.8 1408.09  5415.8 1417.51  5557.9 1422.06
  5725.5 1431.17  5909.9 1455.77  5990.0 1471.65  6035.1 1473.77  6204.5 1495.64
#Mann=7,-1,0
  3901.4    0.05       0  4409.3    0.12       0  4554.9    0.05       0
  4858.9    0.12       0  4982.9    0.07       0  5045.9    0.12       0
  5172.5    0.05       0
Bank Sta=4982.9,5045.9
Exp/Cntr=0.3,0.1

Type RM Length L Ch R = 1,223969,2128,2128,2128
BEGIN DESCRIPTION:
Clear Fork Brazos Rv 58.0
END DESCRIPTION:
XS GIS Cut Line= 4
      1670633.21      7019516.21      1670205.00      7019088.00
      1669705.00      7018588.00      1668705.02      7018088.01
#Sta/Elev= 30
  3677.3 1452.30  4509.2 1416.19  4760.9 1413.68  4919.3 1411.61  4933.4 1406.06
  4947.6 1384.92  4950.0 1384.76  4954.5 1382.76  5004.0 1384.76  5013.7 1389.53
  5034.7 1391.78  5057.1 1386.92  5159.9 1387.17  5177.3 1385.22  5205.2 1399.93
  5249.9 1402.84  5303.0 1432.06  5400.9 1460.24  5429.5 1471.82  5451.2 1482.37
  5563.0 1507.63  5616.1 1523.53  5669.2 1549.64  5719.5 1562.59  5803.4 1592.45
  5876.0 1606.10  5915.2 1619.31  6032.6 1646.47  6071.7 1662.81  6108.0 1668.89
#Mann=7,-1,0
  3677.3    0.05       0  4760.9    0.12       0  4950.0    0.07       0
  5004.0    0.12       0  5013.7    0.05       0  5159.9    0.12       0
  5429.5    0.05       0
Bank Sta=4950,5004
Exp/Cntr=0.3,0.1

Type RM Length L Ch R = 1,221841,1718,1718,1718
BEGIN DESCRIPTION:
Mapping XS 901edd92
END DESCRIPTION:
XS GIS Cut Line= 2
      1671393.34      7019621.86      1671512.65      7017702.16
#Sta/Elev= 30
  3762.9 1466.07  3897.0 1462.11  4227.7 1447.09  4808.8 1413.21  4908.8 1411.77
  4939.0 1411.79  4949.0 1402.55  4959.1 1385.91  4968.3 1382.40  4972.0 1381.40
  5013.3 1382.40  5019.2 1384.58  5039.2 1387.11  5082.4 1385.90  5109.4 1387.93
  5139.4 1385.82  5157.2 1390.84  5189.5 1391.12  5229.6 1405.96  5259.6 1424.09
  5300.3 1444.74  5359.8 1466.12  5379.9 1475.96  5478.7 1514.66  5530.2 1530.64
  5590.3 1544.06  5610.3 1552.51  5639.5 1562.03  5644.5 1562.36  5686.3 1578.12
#Mann=6,-1,0
  3762.9    0.05       0  4908.8    0.12       0  4968.3    0.07       0
  5013.3    0.12       0  5082.4    0.05       0  5300.3    0.12       0
Bank Sta=4968.3,5013.3
Exp/Cntr=0.3,0.1
