HEC-RAS study Fish Creek.prj: Fish Creek Base Level Engineering

--- Fish Creek.g01 (geometry) --- (continued)

Type RM Length L Ch R = 1,63140,436,436,436
BEGIN DESCRIPTION:
Mapping XS 28e11744
END DESCRIPTION:
XS GIS Cut Line= 3
      1679701.89      6984385.08      1679192.82      6984925.33
      1679053.09      6985192.83
#Sta/Elev= 30
  4257.7 1709.20  4394.6 1706.07  4477.2 1703.30  4506.8 1701.89  4561.9 1700.22
  4568.8 1699.40  4674.8 1696.90  4759.7 1695.71  4767.0 1696.37  4773.9 1695.31
  4823.7 1695.08  4915.5 1693.17  4972.1 1690.84  5014.3 1687.00  5024.7 1684.95
  5025.2 1684.45  5033.8 1684.45  5034.3 1684.95  5036.9 1686.43  5045.9 1687.31
  5068.0 1693.89  5082.0 1697.34  5090.1 1698.84  5117.8 1701.62  5128.7 1703.82
  5156.3 1706.06  5184.0 1706.95  5200.5 1708.33  5261.1 1710.33  5301.8 1710.84
#Mann=7,-1,0
  4257.7    0.07       0  4394.6   0.035       0  4477.2    0.07       0
  4506.8   0.035       0  5024.7   0.035       0  5034.3   0.035       0
  5128.7    0.07       0
Bank Sta=5024.7,5034.3
Exp/Cntr=0.3,0.1

Type RM Length L Ch R = 1,62704,675,675,675
BEGIN DESCRIPTION:
Fish Creek 105.0
END DESCRIPTION:
XS GIS Cut Line= 3
      1679666.72      6984406.26      1678849.06      6984679.48
      1678868.63      6985201.52
#Sta/Elev= 30
  4137.9 1708.30  4219.9 1706.61  4231.5 1706.24  4283.7 1704.57  4352.2 1700.91
  4393.2 1699.53  4446.9 1697.76  4631.2 1694.47  4677.4 1694.35  4839.8 1690.43
  4877.8 1689.24  4930.5 1688.77  4941.0 1687.10  4952.4 1683.55  4957.3 1683.11
  4957.8 1682.61  4967.0 1683.11  4984.0 1683.64  5014.1 1686.79  5018.5 1687.07
  5024.3 1688.79  5029.3 1687.62  5038.5 1689.83  5058.6 1691.05  5112.2 1691.70
  5268.7 1693.98  5328.7 1698.03  5378.8 1699.83  5446.5 1705.44  5522.4 1708.43
#Mann=10,-1,0
  4137.9    0.07       0  4219.9   0.035       0  4231.5    0.07       0
  4393.2   0.035       0  4839.8    0.07       0  4957.3    0.07       0
  4967.0    0.07       0  5014.1   0.035       0  5112.2    0.07       0
  5446.5   0.035       0
Bank Sta=4957.3,4967
Exp/Cntr=0.3,0.1

Type RM Length L Ch R = 1,62029,184,184,184
BEGIN DESCRIPTION:
Mapping XS 36b24340
END DESCRIPTION:
XS GIS Cut Line= 5
      1677299.46      6984214.37      1678080.70      6984801.17
      1678427.92      6985051.17      1678511.25      6985085.89
      1678951.10      6985290.23
#Sta/Elev= 30
  3507.4 1735.52  4271.0 1694.66  4364.8 1688.03  4385.6 1685.14  4391.8 1679.98
  4425.4 1679.60  4535.9 1679.92  4542.1 1681.88  4550.6 1689.17  4571.5 1684.57
  4577.7 1680.72  4592.4 1680.06  4678.3 1680.16  4686.9 1687.03  4693.0 1686.73
  4699.3 1681.72  4707.8 1679.20  4713.9 1681.28  4728.6 1679.25  4985.0 1679.13
  4985.5 1678.63  5000.6 1679.13  5048.4 1679.60  5090.1 1682.29  5118.5 1693.64
  5164.3 1696.17  5190.1 1700.71  5307.1 1707.65  5476.3 1711.31  5487.6 1711.94
#Mann=7,-1,0
  3507.4   0.035       0  4425.4   0.033       0  4985.0   0.033       0
  5000.6   0.033       0  5048.4   0.035       0  5190.1    0.07       0
  5476.3   0.035       0
Bank Sta=4985,5000.6
Exp/Cntr=0.3,0.1

Type RM Length L Ch R = 1,61845,168,168,168
BEGIN DESCRIPTION:
Mapping XS c5c66d9c
END DESCRIPTION:
XS GIS Cut Line= 4
      1677302.89      6984440.04      1677868.89      6984822.00
      1678365.42      6985186.59      1678917.47      6985519.90
#Sta/Elev= 30
  3707.7 1729.32  3765.6 1726.96  3858.5 1716.49  4004.6 1710.84  4121.9 1704.91
  4197.0 1700.41  4197.5 1699.91  4212.8 1700.41  4218.3 1701.27  4371.1 1706.11
  4663.7 1707.23  4678.3 1705.36  4699.2 1707.45  4728.5 1705.39  4764.0 1707.54
  4778.7 1705.09  4799.5 1707.70  4814.2 1704.90  4820.4 1707.16  4828.8 1705.39
  4849.7 1707.89  4864.3 1704.60  4904.8 1706.94  4985.3 1706.89  5003.2 1706.86
  5268.9 1700.81  5410.9 1707.54  5540.7 1711.79  5582.1 1712.51  5651.4 1713.87
#Mann=13,-1,0
  3707.7    0.07       0  4004.6   0.035       0  4121.9    0.07       0
  4197.0   0.035       0  4212.8    0.07       0  4218.3   0.035       0
  4904.8    0.07       0  4985.3   0.035       0  5003.2    0.07       0
  5268.9   0.035       0  5410.9    0.07       0  5540.7   0.035       0
  5582.1    0.07       0
Bank Sta=4197,4212.8
Exp/Cntr=0.3,0.1

Type RM Length L Ch R = 1,61677,878,878,878
BEGIN DESCRIPTION:
Mapping XS aac55812
END DESCRIPTION:
XS GIS Cut Line= 5
      1677153.63      6984585.90      1677518.20      6984818.53
      1677868.89      6985006.03      1678223.06      6985269.92
      1678789.00      6985801.14
#Sta/Elev= 30
  3728.3 1727.38  3781.0 1723.63  3796.2 1720.41  3838.5 1716.34  3958.9 1709.40
  4035.7 1705.46  4041.6 1703.71  4056.8 1704.67  4078.0 1702.59  4188.6 1701.07
  4260.0 1698.19  4276.2 1699.24  4299.8 1695.85  4310.5 1695.01  4424.2 1690.14
  4555.2 1686.37  4765.1 1686.39  4902.6 1683.54  4936.1 1682.94  4949.1 1680.35
  4949.6 1679.85  4964.9 1680.35  4965.1 1682.02  4992.4 1683.08  5035.4 1689.56
  5060.5 1690.18  5325.6 1698.84  5530.7 1702.17  5615.7 1705.46  5776.3 1708.45
#Mann=10,-1,0
  3728.3    0.07       0  3958.9   0.035       0  4188.6    0.07       0
  4299.8   0.035       0  4310.5    0.07       0  4424.2   0.035       0
  4902.6    0.07       0  4949.1    0.07       0  4964.9    0.07       0
  5060.5   0.035       0
Bank Sta=4949.1,4964.9
Exp/Cntr=0.3,0.1

Type RM Length L Ch R = 1,60799,537,537,537
BEGIN DESCRIPTION:
Mapping XS a516750e
END DESCRIPTION:
XS GIS Cut Line= 3
      1676551.03      6985603.02      1677498.99      6985641.21
      1678794.11      6985981.49
#Sta/Elev= 30
  4046.0 1753.05  4110.0 1746.66  4180.1 1745.64  4203.3 1741.23  4240.1 1736.24
  4356.6 1728.19  4400.4 1726.01  4500.3 1721.74  4590.4 1715.20  4705.0 1712.17
  4818.1 1706.71  4930.7 1700.03  4970.7 1688.97  4990.2 1679.96  4994.7 1679.96
  4998.8 1676.92  5013.6 1672.92  5014.1 1672.42  5029.6 1672.92  5036.7 1676.30
  5079.5 1682.05  5299.3 1683.74  5523.8 1684.74  5525.0 1684.75  5530.7 1684.76
  5830.7 1689.05  5906.3 1692.48  6183.6 1698.79  6299.5 1706.59  6333.8 1706.87
#Mann=13,-1,0
  4046.0   0.035       0  4203.3    0.07       0  4356.6   0.035       0
  4400.4    0.07       0  4705.0   0.035       0  4818.1    0.07       0
  5013.6    0.07       0  5029.6    0.07       0  5036.7   0.035       0
  5299.3    0.07       0  5523.8   0.035       0  5525.0    0.07       0
  5530.7   0.035       0
Bank Sta=5013.6,5029.6
Exp/Cntr=0.3,0.1

Type RM Length L Ch R = 1,60262,366,366,366
BEGIN DESCRIPTION:
Mapping XS 64c5d829
END DESCRIPTION:
XS GIS Cut Line= 3
      1676519.83      6986207.19      1677710.79      6986092.60
      1678887.89      6986134.27
#Sta/Elev= 30
  3802.0 1720.04  3967.9 1719.43  4223.0 1715.05  4265.5 1714.39  4531.9 1707.51
  4801.8 1700.93  4882.1 1697.68  4912.3 1692.94  4922.3 1689.79  4942.4 1685.65
  4972.6 1674.72  4983.0 1671.96  4983.5 1671.46  4999.0 1671.96  5042.7 1673.57
  5052.7 1674.41  5072.7 1678.70  5102.7 1680.60  5447.0 1683.15  5653.1 1686.20
  5683.1 1687.93  5773.2 1690.35  5843.2 1693.85  5933.3 1696.00  5983.3 1698.29
  6043.3 1702.91  6113.4 1706.01  6139.4 1706.68  6144.4 1705.99  6176.3 1708.96
#Mann=7,-1,0
  3802.0   0.035       0  4223.0    0.07       0  4265.5   0.035       0
  4531.9    0.07       0  4983.0    0.07       0  4999.0    0.07       0
  5447.0   0.035       0
Bank Sta=4983,4999
Exp/Cntr=0.3,0.1

Type RM Length L Ch R = 1,59896,572,572,572
BEGIN DESCRIPTION:
Mapping XS 5db4fde5
END DESCRIPTION:
XS GIS Cut Line= 3
      1677173.78      6986694.72      1677909.85      6986385.70
      1678909.84      6986246.82
#Sta/Elev= 30
  4202.5 1702.27  4467.4 1701.78  4475.0 1702.45  4615.4 1700.74  4620.8 1701.62
  4693.3 1700.18  4789.5 1698.32  4821.8 1697.25  4843.7 1695.21  4897.9 1688.28
  4941.3 1674.00  4980.6 1675.23  5026.2 1675.15  5046.4 1674.88  5058.5 1673.58
  5059.0 1673.08  5074.6 1673.58  5076.7 1674.88  5097.5 1678.74  5213.7 1680.07
  5450.2 1682.78  5599.3 1686.40  5671.0 1689.10  5692.5 1691.32  5711.7 1691.01
  5783.4 1691.80  5803.6 1695.01  5930.4 1703.46  5985.3 1705.86  6010.4 1705.69
#Mann=7,-1,0
  4202.5   0.035       0  4693.3    0.07       0  5058.5    0.07       0
  5074.6    0.07       0  5213.7   0.035       0  5711.7    0.07       0
  5930.4   0.035       0
Bank Sta=5058.5,5074.6
Exp/Cntr=0.3,0.1

Type RM Length L Ch R = 1,59324,951,951,951
BEGIN DESCRIPTION:
Mapping XS 378cecc6
END DESCRIPTION:
XS GIS Cut Line= 3
      1677741.46      6987191.25      1678178.95      6986863.13
      1678937.60      6986368.36
#Sta/Elev= 30
  4452.3 1690.97  4691.6 1689.97  4749.9 1689.18  4799.9 1687.43  4814.5 1685.72
  4820.8 1686.06  4864.5 1680.09  4870.8 1680.26  4906.7 1677.84  4943.7 1676.86
  4964.5 1675.21  4985.4 1671.98  4985.5 1670.66  4986.0 1670.16  5001.6 1670.66
  5021.0 1671.33  5030.2 1672.41  5042.2 1672.45  5057.2 1673.82  5136.9 1676.96
  5304.8 1678.01  5497.8 1683.84  5615.3 1686.40  5686.9 1689.87  5709.1 1692.28
  5736.1 1694.02  5808.6 1697.63  5838.8 1700.78  5875.0 1703.06  5904.9 1704.05
#Mann=5,-1,0
  4452.3   0.035       0  4691.6    0.07       0  4985.5    0.07       0
  5001.6    0.07       0  5136.9   0.035       0
Bank Sta=4985.5,5001.6
Exp/Cntr=0.3,0.1

Type RM Length L Ch R = 1,58373,490,490,490
BEGIN DESCRIPTION:
Mapping XS aa6765fe
END DESCRIPTION:
XS GIS Cut Line= 3
      1677985.10      6987100.44      1678654.34      6987532.71
      1679002.62      6987783.52
#Sta/Elev= 30
  4202.6 1688.30  4254.6 1686.01  4286.4 1683.18  4316.7 1678.69  4331.9 1678.02
  4727.8 1673.46  4779.3 1673.39  4815.5 1674.52  4883.7 1674.12  4916.8 1674.22
  4945.5 1672.50  4960.7 1667.44  4975.9 1666.87  4979.8 1665.71  4980.3 1665.21
  4996.5 1665.71  5017.8 1666.72  5024.8 1671.68  5032.5 1673.74  5038.6 1673.62
  5047.2 1675.33  5068.1 1676.40  5103.7 1676.05  5154.0 1679.62  5168.7 1682.22
  5183.4 1683.63  5260.8 1688.45  5340.5 1696.01  5420.1 1698.91  5428.5 1699.24
#Mann=6,-1,0
  4202.6    0.07       0  4254.6   0.035       0  4883.7    0.07       0
  4979.8    0.07       0  4996.5    0.07       0  5420.1   0.035       0
Bank Sta=4979.8,4996.5
Exp/Cntr=0.3,0.1

Type RM Length L Ch R = 1,57883,368,368,368
BEGIN DESCRIPTION:
Mapping XS 806dcebc
END DESCRIPTION:
XS GIS Cut Line= 3
      1677789.67      6987325.59      1678430.29      6987912.40
      1678667.80      6988153.37
#Sta/Elev= 30
  4131.3 1688.82  4186.3 1687.93  4243.1 1685.68  4278.2 1682.90  4314.0 1681.10
  4355.9 1676.50  4398.5 1675.03  4497.7 1673.49  4518.7 1673.73  4554.5 1672.46
  4611.2 1672.91  4745.6 1670.85  4892.4 1671.84  4943.6 1670.61  4957.8 1669.71
  4979.3 1669.84  5007.4 1666.38  5021.5 1666.14  5027.3 1665.47  5027.8 1664.97
  5043.6 1664.97  5044.1 1665.47  5049.8 1670.83  5064.0 1673.92  5106.3 1679.68
  5162.9 1685.67  5177.0 1688.27  5212.4 1693.26  5290.2 1698.09  5338.4 1699.31
#Mann=4,-1,0
  4131.3   0.035       0  4892.4    0.07       0  5027.3    0.07       0
  5044.1    0.07       0
Bank Sta=5027.3,5044.1
Exp/Cntr=0.3,0.1

Type RM Length L Ch R = 1,57515,528,528,528
BEGIN DESCRIPTION:
Mapping XS 3a553bf0
END DESCRIPTION:
XS GIS Cut Line= 3
      1677454.58      6987525.22      1678110.85      6988035.66
      1678590.02      6988311.70
#Sta/Elev= 30
  4171.6 1688.11  4261.6 1685.13  4359.6 1680.01  4544.2 1674.61  4672.7 1672.95
  4780.2 1670.55  4896.9 1670.65  4957.6 1670.42  4965.0 1668.24  4971.1 1664.98
  4971.6 1664.48  4987.9 1664.98  5000.3 1665.39  5002.5 1666.30  5030.9 1666.89
  5037.2 1666.74  5043.0 1665.48  5053.0 1665.68  5065.5 1668.11  5096.1 1670.29
  5204.6 1669.85  5233.6 1670.81  5250.2 1672.13  5278.6 1678.29  5307.9 1682.84
  5337.5 1684.78  5365.6 1688.03  5417.9 1692.12  5533.8 1696.00  5556.0 1696.71
#Mann=8,-1,0
  4171.6    0.07       0  4261.6   0.035       0  4896.9    0.07       0
  4971.1    0.07       0  4987.9    0.07       0  5204.6   0.035       0
  5233.6    0.07       0  5533.8   0.035       0
Bank Sta=4971.1,4987.9
Exp/Cntr=0.3,0.1

Type RM Length L Ch R = 1,56987,582,582,582
BEGIN DESCRIPTION:
Mapping XS 20154408
END DESCRIPTION:
XS GIS Cut Line= 3
      1677257.58      6987983.68      1678096.16      6988496.73
      1678588.38      6988606.11
#Sta/Elev= 30
  4017.6 1684.83  4113.2 1681.96  4155.8 1678.46  4208.0 1676.13  4223.4 1674.78
  4331.1 1671.76  4476.9 1668.78  4534.2 1668.40  4565.6 1668.01  4729.4 1668.99
  4808.1 1669.21  4898.7 1668.95  4950.9 1666.70  4964.1 1666.84  4972.2 1666.30
  4993.5 1661.06  5000.7 1661.80  5001.3 1660.75  5001.8 1660.25  5017.6 1660.25
  5018.1 1660.75  5020.0 1662.37  5032.5 1668.37  5050.7 1674.99  5081.4 1682.74
  5112.2 1684.74  5198.8 1687.39  5425.7 1692.74  5481.0 1695.19  5504.9 1695.63
#Mann=8,-1,0
  4017.6   0.035       0  4534.2    0.07       0  4729.4   0.035       0
  4808.1    0.07       0  5001.3    0.07       0  5018.1    0.07       0
  5198.8   0.035       0  5425.7    0.07       0
Bank Sta=5001.3,5018.1
Exp/Cntr=0.3,0.1

Type RM Length L Ch R = 1,56405,875,875,875
BEGIN DESCRIPTION:
Mapping XS 0d18b7ee
END DESCRIPTION:
XS GIS Cut Line= 3
      1677067.50      6988171.19      1677783.66      6988965.48
      1678439.86      6988900.38
#Sta/Elev= 30
  3934.6 1685.00  3941.2 1684.86  4049.9 1684.15  4118.1 1683.43  4220.9 1678.67
  4263.5 1675.37  4304.3 1670.06  4369.7 1668.56  4535.7 1667.44  4565.5 1667.32
  4815.8 1665.44  4937.8 1665.77  4971.3 1663.21  4978.7 1663.57  4992.9 1661.08
  5007.0 1660.25  5007.5 1659.75  5023.9 1660.25  5035.6 1660.72  5055.7 1663.61
  5075.8 1662.35  5085.8 1663.61  5105.9 1668.66  5130.7 1672.38  5136.1 1674.19
  5146.1 1675.17  5186.3 1678.46  5234.6 1680.66  5337.5 1683.59  5663.5 1686.58
#Mann=11,-1,0
  3934.6   0.035       0  3941.2    0.07       0  4049.9   0.035       0
  4118.1    0.07       0  4304.3   0.035       0  4535.7    0.07       0
  4565.5   0.035       0  4937.8    0.07       0  5007.0    0.07       0
  5023.9    0.07       0  5234.6   0.035       0
Bank Sta=5007,5023.9
Exp/Cntr=0.3,0.1

Type RM Length L Ch R = 1,55530,664,664,664
BEGIN DESCRIPTION:
Mapping XS 2e6f06a5
END DESCRIPTION:
XS GIS Cut Line= 3
      1676708.15      6989710.26      1677278.45      6989520.16
      1678467.99      6988952.72
#Sta/Elev= 30
  4392.6 1692.10  4568.4 1686.31  4631.7 1686.11  4668.8 1686.99  4795.1 1681.20
  4821.4 1677.74  4858.3 1674.78  4863.6 1673.20  4921.6 1669.81  4947.9 1662.12
  4953.2 1662.81  4958.5 1658.16  4969.0 1654.76  4975.9 1653.71  4976.4 1653.21
  4993.8 1653.71  5008.5 1658.58  5014.0 1659.37  5059.4 1662.55  5414.7 1664.02
  5622.5 1665.37  5699.0 1665.63  5728.6 1666.94  5787.7 1676.09  5842.0 1680.64
  5943.9 1682.78  6028.3 1682.43  6193.8 1683.01  6206.1 1683.44  6311.7 1685.77
#Mann=9,-1,0
  4392.6   0.035       0  4668.8    0.07       0  4975.9    0.07       0
  4993.8    0.07       0  5414.7   0.035       0  5622.5    0.07       0
  6028.3   0.035       0  6193.8    0.07       0  6206.1   0.035       0
Bank Sta=4975.9,4993.8
Exp/Cntr=0.3,0.1

Type RM Length L Ch R = 1,54866,727,727,727
BEGIN DESCRIPTION:
Mapping XS 29724cef
END DESCRIPTION:
XS GIS Cut Line= 3
      1677015.22      6990294.75      1677785.61      6989841.20
      1678780.83      6989418.39
#Sta/Elev= 30
  4097.8 1683.96  4341.0 1676.13  4365.5 1674.34  4453.8 1669.00  4598.6 1666.09
  4620.2 1665.56  4855.4 1662.70  4943.8 1660.44  4956.3 1657.64  4965.3 1657.98
  4971.1 1654.92  4986.8 1655.46  4990.0 1652.75  5001.1 1652.48  5001.6 1651.98
  5019.1 1652.48  5139.2 1655.17  5168.3 1658.46  5175.8 1656.94  5230.2 1660.77
  5343.9 1660.87  5468.4 1662.28  5490.9 1660.81  5534.4 1664.24  5606.7 1665.29
  5686.5 1667.53  5732.1 1675.05  5825.1 1680.25  5849.5 1680.76  6073.1 1691.28
#Mann=12,-1,0
  4097.8   0.035       0  4341.0    0.07       0  4365.5   0.035       0
  4598.6    0.07       0  4620.2   0.035       0  4855.4    0.07       0
  5001.1    0.07       0  5019.1    0.07       0  5343.9   0.035       0
  5606.7    0.07       0  5825.1   0.035       0  5849.5    0.07       0
Bank Sta=5001.1,5019.1
Exp/Cntr=0.3,0.1

Type RM Length L Ch R = 1,54139,567,567,567
BEGIN DESCRIPTION:
Mapping XS e2f6a9b7
END DESCRIPTION:
XS GIS Cut Line= 3
      1677091.07      6990435.96      1678203.00      6990279.71
      1678730.83      6990167.91
#Sta/Elev= 30
  3874.7 1679.74  3959.5 1677.04  4100.8 1671.00  4185.0 1669.02  4232.1 1667.02
  4256.3 1667.02  4373.5 1664.19  4546.5 1661.07  4848.1 1658.07  4897.8 1655.58
  4939.0 1654.87  4959.2 1650.84  4970.3 1649.45  4970.8 1648.95  4988.0 1648.95
  4988.5 1649.45  4993.9 1652.13  4996.0 1653.10  5001.1 1653.10  5009.8 1657.44
  5020.0 1661.37  5027.6 1663.56  5032.7 1663.94  5050.7 1668.83  5082.3 1672.49
  5214.3 1675.81  5296.0 1680.25  5408.5 1683.85  5469.5 1687.27  5537.1 1689.78
#Mann=5,-1,0
  3874.7   0.035       0  4970.3    0.07       0  4988.5   0.035       0
  4993.9    0.07       0  5469.5   0.035       0
Bank Sta=4970.3,4988.5
Exp/Cntr=0.3,0.1

Type RM Length L Ch R = 1,53572,494,494,494
BEGIN DESCRIPTION:
Mapping XS e92f4b42
END DESCRIPTION:
XS GIS Cut Line= 3
      1677195.10      6991010.79      1678198.57      6990798.98
      1678881.35      6990719.27
#Sta/Elev= 30
  3969.2 1680.28  4110.7 1673.92  4150.1 1671.00  4155.2 1671.37  4199.8 1669.03
  4510.8 1659.01  4674.3 1656.10  4887.9 1655.62  4899.2 1656.15  4940.0 1655.53
  4950.3 1654.18  4966.5 1649.60  4967.0 1649.10  4984.7 1649.60  4990.4 1650.99
  5001.3 1651.89  5051.6 1652.72  5091.9 1662.39  5129.9 1668.74  5134.9 1668.10
  5142.2 1669.43  5172.4 1670.41  5253.0 1670.37  5306.7 1671.49  5395.1 1675.69
  5468.9 1681.46  5552.9 1684.85  5575.1 1686.23  5615.4 1690.54  5682.2 1693.84
#Mann=7,-1,0
  3969.2    0.07       0  4110.7   0.035       0  4887.9    0.07       0
  4966.5    0.07       0  4984.7    0.07       0  5468.9   0.035       0
  5552.9    0.07       0
Bank Sta=4966.5,4984.7
Exp/Cntr=0.3,0.1

Type RM Length L Ch R = 1,53078,529,529,529
BEGIN DESCRIPTION:
Mapping XS 184ecdb8
END DESCRIPTION:
XS GIS Cut Line= 3
      1677196.73      6991354.25      1678207.98      6991291.31
      1678740.95      6991256.65
#Sta/Elev= 30
  3983.9 1674.17  4045.5 1672.08  4182.6 1669.22  4382.9 1663.42  4433.0 1659.00
  4473.1 1657.63  4503.2 1654.72  4533.2 1653.39  4643.2 1651.09  4924.0 1654.86
  4934.0 1654.42  4944.0 1652.31  4944.9 1648.65  4945.4 1648.15  4963.2 1648.65
  4969.3 1649.55  5024.2 1650.03  5054.2 1652.68  5122.3 1652.13  5127.3 1652.77
  5134.4 1651.85  5184.5 1654.33  5194.5 1655.11  5224.6 1659.98  5279.5 1665.86
  5294.8 1668.75  5344.9 1674.88  5425.0 1680.44  5475.1 1686.88  5531.2 1691.35
#Mann=5,-1,0
  3983.9    0.07       0  4045.5   0.035       0  4944.9    0.07       0
  4963.2   0.035       0  4969.3    0.07       0
Bank Sta=4944.9,4963.2
Exp/Cntr=0.3,0.1

Type RM Length L Ch R = 1,52549,790,790,790
BEGIN DESCRIPTION:
Mapping XS b0fe2e41
END DESCRIPTION:
XS GIS Cut Line= 3
      1677188.00      6991519.18      1678355.55      6991675.43
      1678739.67      6991731.85
#Sta/Elev= 30
  3822.4 1670.27  3838.1 1670.03  4233.1 1662.77  4263.3 1660.92  4270.9 1658.72
  4333.9 1644.55  4370.0 1642.21  4370.5 1641.71  4388.3 1642.21  4419.5 1646.47
  4434.8 1648.84  4466.6 1649.49  4555.9 1646.85  4611.8 1647.26  4663.0 1649.10
  4676.2 1649.18  4681.2 1646.71  4747.6 1649.69  4787.9 1647.90  4838.4 1651.13
  4905.3 1651.89  5002.6 1645.41  5009.9 1649.11  5048.9 1655.36  5080.7 1666.72
  5131.2 1675.04  5193.5 1681.38  5258.2 1690.85  5387.2 1694.16  5388.6 1694.16
#Mann=10,-1,0
  3822.4    0.07       0  3838.1   0.035       0  4270.9    0.07       0
  4370.0    0.07       0  4388.3    0.07       0  4419.5   0.035       0
  4466.6    0.07       0  4611.8   0.035       0  4663.0    0.07       0
  5387.2   0.035       0
Bank Sta=4370,4388.3
Exp/Cntr=0.3,0.1

Type RM Length L Ch R = 1,51759,142,142,142
BEGIN DESCRIPTION:
Fish Creek 85.0
END DESCRIPTION:
XS GIS Cut Line= 4
      1677170.85      6991729.00      1677532.82      6991926.91
      1677715.77      6991928.27      1678579.97      6991963.00
#Sta/Elev= 30
  4404.5 1666.34  4664.3 1660.34  4739.8 1660.49  4827.2 1661.77  4889.2 1661.13
  4899.2 1659.69  4909.2 1653.03  4919.2 1643.45  4929.2 1641.47  4939.2 1640.78
  4988.0 1639.70  4988.5 1639.20  5005.8 1639.20  5006.3 1639.70  5256.2 1640.41
  5330.9 1640.07  5365.7 1640.10  5370.7 1640.71  5459.6 1640.61  5539.7 1642.78
  5559.7 1644.10  5589.7 1651.93  5615.3 1660.38  5669.8 1664.58  5699.8 1668.68
  5719.8 1672.53  5749.8 1677.06  5809.9 1682.38  5829.9 1686.16  5864.9 1688.19
#Mann=6,-1,0
  4404.5   0.035       0  4827.2    0.07       0  4988.0    0.07       0
  5006.3    0.07       0  5256.2   0.035       0  5330.9    0.07       0
Bank Sta=4988,5006.3
Exp/Cntr=0.3,0.1

Type RM Length L Ch R = 1,51617,138,138,138
BEGIN DESCRIPTION:
Mapping XS 1f18fc05
END DESCRIPTION:
XS GIS Cut Line= 4
      1677012.01      6991729.01      1677538.03      6992064.93
      1677702.09      6992067.54      1678524.97      6992080.56
#Sta/Elev= 30
  4208.9 1668.28  4253.7 1666.47  4305.3 1665.84  4326.5 1664.66  4362.9 1664.53
  4384.0 1663.76  4399.2 1664.22  4472.0 1662.79  4635.4 1657.77  4635.9 1657.27
  4653.2 1657.27  4653.7 1657.77  4717.3 1659.48  4790.1 1660.67  4805.3 1661.48
  4817.6 1663.28  4860.0 1665.40  4910.0 1667.18  4959.7 1667.77  5155.1 1668.08
  5261.1 1667.35  5338.7 1666.41  5343.7 1667.52  5480.1 1666.38  5640.1 1663.95
  5700.1 1664.30  5730.1 1666.88  5760.1 1671.59  5800.1 1676.92  5820.1 1678.60
#Mann=6,-1,0
  4208.9   0.035       0  4635.4    0.07       0  4653.7   0.035       0
  4959.7    0.07       0  5155.1   0.035       0  5261.1    0.07       0
Bank Sta=4635.4,4653.7
Exp/Cntr=0.3,0.1

Type RM Length L Ch R = 1,51479,562,562,562
BEGIN DESCRIPTION:
Fish Creek 84.0
END DESCRIPTION:
XS GIS Cut Line= 4
      1676959.88      6991768.05      1677410.21      6992136.16
      1677705.01      6992205.99      1678564.89      6992186.46
#Sta/Elev= 30
  4115.4 1667.96  4175.4 1664.58  4275.9 1663.75  4360.6 1660.01  4389.3 1660.75
  4424.5 1659.13  4438.8 1659.49  4488.4 1656.45  4593.1 1654.78  4694.4 1655.21
  4722.0 1656.69  4727.2 1656.08  4763.6 1657.79  4853.9 1659.63  4876.7 1656.81
  4907.5 1648.69  4928.0 1646.06  4943.5 1645.27  4948.7 1643.68  4979.4 1643.44
  4981.8 1642.26  4982.3 1641.76  5000.1 1642.26  5060.0 1646.85  5139.7 1648.31
  5258.5 1648.99  5640.2 1650.58  5790.2 1658.93  5830.2 1659.87  5860.1 1659.37
#Mann=6,-1,0
  4115.4   0.035       0  4593.1    0.07       0  4981.8    0.07       0
  5000.1    0.07       0  5139.7   0.035       0  5258.5    0.07       0
Bank Sta=4981.8,5000.1
Exp/Cntr=0.3,0.1

Type RM Length L Ch R = 1,50917,798,798,798
BEGIN DESCRIPTION:
Fish Creek 83.0
END DESCRIPTION:
XS GIS Cut Line= 3
      1676530.90      6992181.86      1677605.00      6992738.00
      1678537.85      6993456.16
#Sta/Elev= 30
  3794.6 1673.37  4107.2 1668.64  4171.6 1668.19  4210.3 1665.51  4351.0 1660.35
  4418.0 1659.93  4558.8 1657.46  4625.2 1653.54  4669.5 1647.55  4700.1 1646.26
  4901.7 1645.41  4951.6 1641.63  4964.4 1638.36  4964.9 1637.86  4983.0 1638.36
  5061.2 1644.76  5223.9 1641.99  5260.5 1641.62  5281.8 1639.49  5310.4 1639.76
  5339.4 1644.95  5360.2 1644.94  5403.7 1649.82  5478.2 1651.51  5513.3 1652.68
  5596.7 1655.43  5646.6 1658.65  5688.2 1664.19  5810.5 1676.41  6181.4 1690.56
#Mann=8,-1,0
  3794.6   0.035       0  4107.2    0.07       0  4418.0   0.035       0
  4964.4   0.035       0  4983.0   0.035       0  5223.9    0.07       0
  5478.2   0.035       0  5513.3    0.07       0
Bank Sta=4964.4,4983
Exp/Cntr=0.3,0.1

Type RM Length L Ch R = 1,50119,641,641,641
BEGIN DESCRIPTION:
Mapping XS 32bc9a23
END DESCRIPTION:
XS GIS Cut Line= 3
      1676393.04      6992526.28      1677462.52      6993442.98
      1678201.04      6994160.69
#Sta/Elev= 30
  3595.7 1674.57  3782.7 1667.53  3980.8 1654.54  4002.8 1654.70  4023.6 1652.93
  4158.6 1647.60  4293.6 1644.82  4478.0 1643.07  4662.6 1643.35  4690.9 1643.46
  4746.9 1641.23  4796.8 1642.79  4849.9 1641.75  4881.9 1641.36  4939.0 1637.72
  4951.9 1638.63  5012.3 1636.66  5012.8 1636.16  5035.0 1636.66  5076.1 1639.56
  5108.5 1644.22  5174.3 1647.71  5320.7 1656.48  5462.2 1662.27  5603.7 1672.41
  5610.6 1674.07  5716.8 1676.73  5780.4 1680.60  5865.3 1683.74  6034.1 1687.21
#Mann=8,-1,0
  3595.7   0.035       0  4662.6    0.07       0  4849.9   0.035       0
  4951.9    0.07       0  5012.3    0.07       0  5035.0    0.07       0
  5076.1   0.035       0  5174.3    0.07       0
Bank Sta=5012.3,5035
Exp/Cntr=0.3,0.1

Type RM Length L Ch R = 1,49478,592,592,592
BEGIN DESCRIPTION:
Mapping XS 9c40e3fe
END DESCRIPTION:
XS GIS Cut Line= 3
      1676070.16      6992974.23      1676979.88      6993769.37
      1677871.16      6994365.86
#Sta/Elev= 30
  3797.1 1673.71  3801.1 1673.71  3918.2 1669.01  4157.7 1653.74  4334.8 1650.48
  4384.6 1648.50  4419.7 1648.71  4759.8 1642.02  4933.1 1641.34  4944.6 1640.95
  4958.8 1637.33  4965.5 1634.92  4968.2 1632.11  4968.7 1631.61  4991.1 1632.11
  4993.9 1634.05  5029.7 1636.83  5086.7 1636.49  5131.8 1639.35  5281.9 1641.50
  5354.0 1644.56  5390.0 1647.91  5432.6 1657.78  5492.1 1668.93  5528.1 1671.41
  5570.1 1676.32  5630.5 1679.85  5741.1 1681.22  5801.6 1682.29  6077.8 1688.21
#Mann=9,-1,0
  3797.1   0.035       0  3801.1    0.07       0  3918.2   0.035       0
  4933.1    0.07       0  4968.2    0.07       0  4991.1    0.07       0
  5630.5   0.035       0  5741.1    0.07       0  5801.6   0.035       0
Bank Sta=4968.2,4991.1
Exp/Cntr=0.3,0.1

Type RM Length L Ch R = 1,48886,213,213,213
BEGIN DESCRIPTION:
Mapping XS 0d9fb7a2
END DESCRIPTION:
XS GIS Cut Line= 3
      1675880.35      6993315.90      1676803.96      6994291.59
      1677790.06      6994486.03
#Sta/Elev= 30
  3658.5 1670.31  3662.0 1670.31  3762.2 1670.07  3983.0 1655.36  3993.7 1654.49
  4137.2 1648.06  4448.3 1643.31  4512.2 1639.41  4589.9 1639.85  4632.4 1636.50
  4653.4 1641.14  4823.3 1638.11  4844.8 1634.71  4916.9 1638.79  4957.6 1638.48
  4999.1 1632.94  5042.6 1631.35  5043.1 1630.85  5065.5 1631.35  5074.4 1636.92
  5105.0 1639.63  5298.7 1642.48  5321.8 1645.20  5391.0 1661.66  5419.4 1667.94
  5441.4 1669.38  5555.6 1670.25  5699.6 1672.34  5886.4 1682.35  6007.1 1685.35
#Mann=10,-1,0
  3658.5    0.07       0  3662.0   0.035       0  3983.0    0.07       0
  3993.7   0.035       0  4916.9    0.07       0  5042.6    0.07       0
  5065.5    0.07       0  5391.0   0.035       0  5555.6    0.07       0
  5699.6   0.035       0
Bank Sta=5042.6,5065.5
Exp/Cntr=0.3,0.1

Type RM Length L Ch R = 1,48673,458,458,458
BEGIN DESCRIPTION:
Mapping XS c6af5797
END DESCRIPTION:
XS GIS Cut Line= 3
      1675064.38      6994361.03      1676689.37      6994451.31
      1677910.76      6994694.20
#Sta/Elev= 30
  3370.6 1672.67  3505.0 1670.74  3641.6 1668.28  3801.9 1659.21  3831.9 1661.71
  3862.0 1656.94  4152.4 1646.07  4628.1 1639.16  4653.2 1638.53  4668.1 1635.30
  4671.4 1629.42  4671.9 1628.92  4695.0 1629.42  4703.3 1633.97  4723.3 1635.19
  4743.3 1632.42  4953.7 1635.63  5002.7 1631.42  5034.4 1638.19  5088.1 1638.97
  5177.2 1637.26  5268.4 1639.97  5519.1 1646.93  5728.7 1657.53  5788.9 1656.20
  5855.7 1665.53  5877.0 1670.14  6075.7 1681.18  6120.6 1682.29  6243.4 1686.62
#Mann=10,-1,0
  3370.6    0.07       0  3505.0   0.035       0  4628.1    0.07       0
  4671.4    0.07       0  4695.0    0.07       0  5088.1   0.035       0
  5268.4    0.07       0  5855.7   0.035       0  6075.7    0.07       0
  6120.6   0.035       0
Bank Sta=4671.4,4695
Exp/Cntr=0.3,0.1

Type RM Length L Ch R = 1,48215,482,482,482
BEGIN DESCRIPTION:
Mapping XS 402a487e
END DESCRIPTION:
XS GIS Cut Line= 3
      1675144.28      6994482.57      1676356.04      6994687.42
      1677635.84      6994923.27
#Sta/Elev= 30
  3772.7 1675.48  3824.3 1674.66  3925.6 1672.79  4118.3 1666.77  4194.8 1660.22
  4315.6 1660.21  4444.1 1646.87  4473.2 1644.13  4655.8 1639.53  4929.0 1637.47
  4960.0 1636.78  4975.2 1634.17  4978.6 1629.11  4979.1 1628.61  5002.3 1629.11
  5061.6 1634.73  5102.3 1636.64  5239.2 1637.97  5437.8 1635.51  5474.8 1636.75
  5559.9 1638.36  5619.1 1642.28  5671.7 1652.40  5715.8 1656.12  5836.5 1664.37
  5885.2 1668.89  5971.1 1671.38  6088.6 1678.39  6258.7 1683.35  6303.0 1684.67
#Mann=13,-1,0
  3772.7    0.07       0  3824.3   0.035       0  3925.6    0.07       0
  4444.1   0.035       0  4929.0    0.07       0  4978.6    0.07       0
  5002.3    0.07       0  5239.2   0.035       0  5474.8    0.07       0
  5619.1   0.035       0  5715.8    0.07       0  5836.5   0.035       0
  6258.7    0.07       0
Bank Sta=4978.6,5002.3
Exp/Cntr=0.3,0.1

Type RM Length L Ch R = 1,47733,484,484,484
BEGIN DESCRIPTION:
Mapping XS fc459531
END DESCRIPTION:
XS GIS Cut Line= 3
      1675510.89      6994867.06      1676580.37      6995019.84
      1677309.52      6995075.40
#Sta/Elev= 30
  3912.4 1659.74  3946.9 1658.24  3987.3 1652.30  4078.8 1645.59  4108.5 1642.21
  4165.3 1639.66  4383.9 1636.10  4528.4 1635.35  4704.5 1635.55  4775.2 1630.82
  4795.4 1631.35  4803.8 1634.77  4806.7 1636.28  4877.4 1636.17  4936.8 1633.57
  4943.1 1631.54  4948.2 1635.20  4980.7 1627.93  4981.2 1627.43  5004.4 1627.93
  5087.6 1629.61  5117.7 1628.09  5147.8 1630.66  5169.4 1629.85  5268.2 1645.98
  5320.1 1649.11  5341.7 1650.36  5551.5 1667.38  5619.2 1670.02  5724.0 1677.41
#Mann=10,-1,0
  3912.4    0.07       0  4078.8   0.035       0  4383.9    0.07       0
  4528.4   0.035       0  4803.8    0.07       0  4980.7    0.07       0
  5004.4    0.07       0  5320.1   0.035       0  5341.7    0.07       0
  5551.5   0.035       0
Bank Sta=4980.7,5004.4
Exp/Cntr=0.3,0.1

Type RM Length L Ch R = 1,47249,338,338,338
BEGIN DESCRIPTION:
Mapping XS 617921a9
END DESCRIPTION:
XS GIS Cut Line= 3
      1675486.34      6995053.27      1676480.26      6995417.85
      1677100.43      6995534.94
#Sta/Elev= 30
  3944.9 1658.75  3955.0 1658.25  4002.1 1655.68  4032.6 1650.74  4051.1 1650.40
  4118.8 1648.98  4135.2 1642.30  4167.2 1639.54  4316.3 1633.72  4486.7 1633.45
  4508.0 1631.73  4591.7 1633.78  4641.1 1634.06  4657.1 1635.80  4689.1 1634.00
  4742.3 1635.23  4847.2 1634.00  4912.8 1633.24  4960.6 1627.55  4979.1 1628.45
  5006.7 1626.56  5007.2 1626.06  5030.5 1626.56  5049.1 1627.11  5085.0 1636.88
  5357.1 1648.73  5486.7 1657.55  5557.9 1665.32  5597.9 1666.94  5634.7 1670.25
#Mann=9,-1,0
  3944.9   0.035       0  3955.0    0.07       0  4051.1   0.035       0
  4591.7    0.07       0  4847.2   0.035       0  4979.1    0.07       0
  5006.7    0.07       0  5030.5    0.07       0  5597.9   0.035       0
Bank Sta=5006.7,5030.5
Exp/Cntr=0.3,0.1

Type RM Length L Ch R = 1,46911,411,411,411
BEGIN DESCRIPTION:
Mapping XS e01623ce
END DESCRIPTION:
XS GIS Cut Line= 3
      1675304.09      6995437.39      1676245.88      6995643.54
      1677077.09      6995791.12
#Sta/Elev= 30
  4035.4 1664.66  4056.7 1664.08  4138.7 1657.45  4198.5 1655.96  4247.4 1649.53
  4266.5 1648.11  4340.3 1639.91  4438.2 1633.34  4589.1 1632.53  4732.4 1633.46
  4760.6 1632.49  4793.9 1632.62  4809.6 1633.91  4937.2 1634.11  4967.9 1632.65
  4978.1 1630.96  4986.3 1625.00  4986.8 1624.50  5010.1 1625.00  5018.9 1627.88
  5029.1 1628.80  5049.0 1628.51  5108.0 1625.30  5191.6 1632.69  5384.1 1635.25
  5465.8 1637.43  5511.4 1639.89  5683.5 1655.24  5760.3 1664.03  5843.7 1669.29
#Mann=5,-1,0
  4035.4    0.07       0  4266.5   0.035       0  4986.3   0.035       0
  5010.1   0.035       0  5384.1    0.07       0
Bank Sta=4986.3,5010.1
Exp/Cntr=0.3,0.1

Type RM Length L Ch R = 1,46500,640,640,640
BEGIN DESCRIPTION:
Mapping XS a25c8554
END DESCRIPTION:
XS GIS Cut Line= 3
      1675139.95      6996295.32      1676103.52      6996008.85
      1677064.91      6995945.91
#Sta/Elev= 30
  3993.5 1663.76  4100.5 1661.70  4199.6 1658.65  4311.5 1650.53  4317.2 1646.65
  4363.9 1644.19  4415.7 1644.65  4427.2 1643.64  4436.9 1639.42  4541.3 1629.66
  4592.3 1628.93  4656.0 1628.24  4833.4 1631.47  4870.9 1627.68  4951.2 1627.13
  4989.9 1624.98  4998.4 1622.90  4998.9 1622.40  5022.2 1622.90  5040.3 1624.80
  5060.4 1623.60  5086.9 1628.34  5146.6 1630.30  5330.9 1630.43  5540.5 1634.64
  5641.6 1639.57  5721.8 1649.71  5850.4 1663.01  5892.1 1664.56  5962.2 1670.06
#Mann=11,-1,0
  3993.5    0.07       0  4100.5   0.035       0  4199.6    0.07       0
  4311.5   0.035       0  4415.7    0.07       0  4592.3   0.035       0
  4870.9    0.07       0  4998.4    0.07       0  5022.2    0.07       0
  5146.6   0.035       0  5540.5    0.07       0
Bank Sta=4998.4,5022.2
Exp/Cntr=0.3,0.1

Type RM Length L Ch R = 1,45860,903,903,903
BEGIN DESCRIPTION:
Mapping XS 1ffa4a60
END DESCRIPTION:
XS GIS Cut Line= 3
      1675265.89      6996948.50      1676381.30      6996369.09
      1677019.01      6996122.65
#Sta/Elev= 30
  3738.4 1663.71  3741.6 1663.67  3827.6 1660.22  3924.2 1652.41  3967.8 1651.02
  4028.5 1643.22  4074.7 1640.92  4311.0 1633.55  4318.3 1633.68  4570.2 1625.80
  4680.7 1625.31  4725.0 1623.14  4769.2 1627.53  4801.8 1627.90  4910.7 1627.66
  4940.5 1626.84  5019.6 1619.33  5020.1 1618.83  5043.4 1619.33  5043.8 1621.24
  5052.9 1624.14  5074.3 1627.46  5160.1 1631.33  5239.3 1631.99  5299.8 1633.62
  5430.9 1641.44  5505.5 1652.44  5578.2 1661.15  5652.2 1664.33  5679.0 1666.98
#Mann=14,-1,0
  3738.4    0.07       0  3741.6   0.035       0  3924.2    0.07       0
  4074.7   0.035       0  4311.0    0.07       0  4318.3   0.035       0
  4801.8    0.07       0  4910.7   0.035       0  5019.6   0.035       0
  5043.4   0.035       0  5239.3   0.035       0  5299.8    0.07       0
  5505.5   0.035       0  5652.2    0.07       0
Bank Sta=5019.6,5043.4
Exp/Cntr=0.3,0.1

Type RM Length L Ch R = 1,44957,705,705,705
BEGIN DESCRIPTION:
Mapping XS 6a2b065a
END DESCRIPTION:
XS GIS Cut Line= 3
      1675451.57      6997369.83      1676104.82      6997074.68
      1677109.59      6996456.19
#Sta/Elev= 30
  4283.3 1662.68  4414.9 1659.03  4469.0 1656.63  4506.5 1652.79  4561.4 1650.59
  4649.2 1636.07  4725.9 1632.01  4945.5 1625.15  5004.8 1618.82  5012.1 1617.34
  5014.0 1615.07  5014.5 1614.57  5038.2 1615.07  5041.5 1618.96  5062.0 1620.98
  5084.4 1621.23  5136.1 1624.82  5352.6 1625.11  5536.1 1630.10  5578.6 1629.73
  5636.6 1631.73  5657.0 1630.93  5752.5 1632.06  5804.6 1636.12  5820.0 1639.81
  5841.3 1642.43  5978.5 1650.45  6125.3 1656.67  6131.2 1658.10  6180.0 1659.35
#Mann=8,-1,0
  4283.3   0.035       0  4414.9    0.07       0  4725.9   0.035       0
  5014.0   0.035       0  5038.2   0.035       0  5062.0    0.07       0
  5084.4   0.035       0  5657.0    0.07       0
Bank Sta=5014,5038.2
Exp/Cntr=0.3,0.1

Type RM Length L Ch R = 1,44252,541,541,541
BEGIN DESCRIPTION:
Mapping XS 43fe0c2a
END DESCRIPTION:
XS GIS Cut Line= 3
      1675737.56      6997848.14      1676210.62      6997746.15
      1677711.21      6997531.47
#Sta/Elev= 30
  4513.0 1652.68  4586.0 1654.04  4728.8 1651.58  4745.7 1649.23  4789.3 1639.02
  4848.0 1627.10  4866.4 1621.29  4873.6 1621.06  4893.2 1620.87  4929.8 1622.00
  4965.0 1619.38  4968.8 1617.11  4969.3 1616.61  4993.0 1617.11  4996.6 1618.79
  5072.1 1618.74  5088.5 1621.11  5102.4 1621.03  5132.7 1617.55  5152.9 1621.02
  5183.2 1622.26  5546.9 1625.32  5789.3 1632.08  5849.9 1634.51  5865.8 1636.48
  6193.4 1645.77  6308.2 1650.91  6395.4 1653.93  6462.4 1658.49  6512.8 1661.54
#Mann=8,-1,0
  4513.0    0.07       0  4789.3   0.035       0  4873.6    0.07       0
  4893.2   0.035       0  4968.8   0.035       0  4993.0   0.035       0
  6308.2    0.07       0  6462.4   0.035       0
Bank Sta=4968.8,4993
Exp/Cntr=0.3,0.1

Type RM Length L Ch R = 1,43711,227,227,227
BEGIN DESCRIPTION:
Mapping XS 65459006
END DESCRIPTION:
XS GIS Cut Line= 3
      1675752.79      6997945.26      1676302.27      6998190.06
      1677557.43      6998096.31
#Sta/Elev= 30
  4396.1 1642.79  4415.0 1643.62  4420.5 1642.21  4438.3 1642.38  4467.0 1640.44
  4484.7 1640.43  4490.2 1639.49  4583.1 1636.99  4628.4 1634.08  4672.2 1627.12
  4712.3 1623.73  4792.6 1617.08  4831.9 1620.69  4907.1 1620.73  4959.0 1619.05
  4976.8 1616.38  4977.4 1615.35  4977.9 1614.85  5001.9 1615.35  5007.1 1615.62
  5060.5 1620.57  5069.3 1620.43  5089.0 1621.14  5431.6 1621.28  5754.0 1630.28
  5882.8 1634.27  5983.1 1638.73  6103.4 1647.67  6162.5 1655.26  6256.3 1661.32
#Mann=7,-1,0
  4396.1    0.07       0  4712.3   0.035       0  4977.4   0.035       0
  5001.9   0.035       0  5007.1    0.07       0  5069.3   0.035       0
  5754.0    0.07       0
Bank Sta=4977.4,5001.9
Exp/Cntr=0.3,0.1

Type RM Length L Ch R = 1,43484,328,328,328
BEGIN DESCRIPTION:
Mapping XS 3d01c6b3
END DESCRIPTION:
XS GIS Cut Line= 3
      1675156.41      6998408.81      1676260.60      6998400.99
      1677611.04      6998286.51
#Sta/Elev= 30
  3900.4 1658.74  3999.0 1653.25  4079.0 1651.03  4139.0 1643.52  4179.0 1639.95
  4257.5 1636.14  4294.0 1634.58  4579.0 1620.69  4689.0 1621.28  4759.0 1619.59
  4939.0 1618.60  5026.7 1614.09  5027.2 1613.59  5051.5 1614.09  5059.2 1617.99
  5079.3 1620.14  5216.0 1620.30  5240.1 1620.25  5400.4 1620.21  5551.0 1621.85
  5721.6 1624.44  5853.4 1628.59  5922.3 1630.99  6047.0 1638.00  6113.0 1646.02
  6166.4 1650.45  6183.2 1653.36  6273.5 1660.30  6303.7 1664.53  6359.9 1669.23
#Mann=8,-1,0
  3900.4   0.035       0  4257.5    0.07       0  4294.0   0.035       0
  5026.7   0.035       0  5051.5   0.035       0  5216.0    0.07       0
  5240.1   0.035       0  5853.4    0.07       0
Bank Sta=5026.7,5051.5
Exp/Cntr=0.3,0.1

Type RM Length L Ch R = 1,43156,321,321,321
BEGIN DESCRIPTION:
Mapping XS bd62a572
END DESCRIPTION:
XS GIS Cut Line= 3
      1675171.40      6998923.03      1676106.26      6998670.44
      1677624.48      6998498.56
#Sta/Elev= 30
  4033.8 1659.19  4038.3 1658.08  4067.8 1658.32  4083.0 1656.95  4222.2 1654.10
  4267.3 1651.45  4336.7 1649.78  4410.4 1638.78  4483.5 1632.48  4793.7 1622.50
  4879.6 1618.08  4897.3 1618.10  4928.4 1615.49  4938.7 1613.26  4967.7 1612.90
  4968.2 1612.40  4992.6 1612.90  5021.0 1614.93  5061.3 1614.60  5151.9 1618.99
  5421.2 1619.19  5511.0 1617.88  5614.8 1620.26  5836.2 1622.50  5994.0 1626.04
  6107.9 1630.18  6178.4 1634.27  6269.0 1641.91  6419.9 1656.66  6530.1 1662.53
#Mann=6,-1,0
  4033.8   0.035       0  4083.0    0.07       0  4483.5   0.035       0
  4967.7   0.035       0  4992.6   0.035       0  5994.0    0.07       0
Bank Sta=4967.7,4992.6
Exp/Cntr=0.3,0.1

Type RM Length L Ch R = 1,42835,321,321,321
BEGIN DESCRIPTION:
Mapping XS 1ff15bdf
END DESCRIPTION:
XS GIS Cut Line= 3
      1675231.96      6998999.95      1676004.53      6998960.02
      1677081.28      6999116.07
#Sta/Elev= 30
  4225.9 1661.45  4283.1 1661.40  4379.1 1659.96  4459.3 1655.83  4519.3 1649.72
  4579.4 1638.72  4661.7 1631.46  4929.9 1621.20  4959.9 1618.65  4990.0 1611.48
  4995.5 1611.33  4997.6 1610.99  4998.1 1610.49  5022.5 1610.99  5022.8 1612.44
  5040.4 1613.33  5111.1 1618.16  5303.7 1615.60  5545.6 1616.19  5579.5 1615.54
  5606.2 1612.98  5636.6 1615.94  5737.6 1617.06  5785.1 1616.64  5828.5 1613.89
  5879.1 1615.64  5925.6 1621.15  6020.5 1628.97  6059.8 1630.94  6087.5 1631.48
#Mann=8,-1,0
  4225.9   0.035       0  4283.1    0.07       0  4661.7   0.035       0
  4995.5    0.07       0  4997.6    0.07       0  5022.5    0.07       0
  5040.4   0.035       0  6059.8    0.07       0
Bank Sta=4997.6,5022.5
Exp/Cntr=0.3,0.1

Type RM Length L Ch R = 1,42514,266,266,266
BEGIN DESCRIPTION:
Mapping XS c108f179
END DESCRIPTION:
XS GIS Cut Line= 3
      1675392.76      6999298.04      1675900.53      6999232.94
      1677015.10      6999292.83
#Sta/Elev= 30
  4486.3 1662.76  4529.9 1662.13  4579.3 1659.19  4660.0 1648.16  4710.4 1639.78
  4815.1 1627.90  4861.6 1623.22  4901.9 1620.99  4918.1 1617.67  4923.1 1619.47
  4960.1 1613.78  4972.5 1611.73  5012.7 1612.50  5022.7 1610.60  5032.7 1610.64
  5052.8 1614.58  5080.1 1616.51  5243.0 1617.31  5463.4 1614.41  5483.4 1613.26
  5491.0 1610.40  5491.5 1609.90  5515.9 1610.40  5553.5 1614.18  5573.5 1614.75
  5768.6 1614.74  5884.0 1610.92  5981.7 1621.68  6044.2 1632.44  6114.4 1633.59
#Mann=8,-1,0
  4486.3    0.07       0  4815.1   0.035       0  4960.1    0.07       0
  5080.1   0.035       0  5491.0    0.07       0  5515.9   0.035       0
  5768.6    0.07       0  5981.7   0.035       0
Bank Sta=5491,5515.9
Exp/Cntr=0.3,0.1

Type RM Length L Ch R = 1,42248,463,463,463
BEGIN DESCRIPTION:
Mapping XS 42644b85
END DESCRIPTION:
XS GIS Cut Line= 3
      1675257.27      6999607.95      1675801.58      6999467.31
      1676981.94      6999430.91
#Sta/Elev= 30
  4434.8 1662.00  4608.7 1659.87  4695.1 1659.32  4735.8 1657.11  4771.2 1651.55
  4817.1 1647.32  4944.8 1627.95  4974.5 1623.64  4990.2 1618.88  4996.2 1614.70
  5004.9 1613.27  5020.4 1607.83  5070.4 1612.94  5125.5 1614.66  5380.6 1616.09
  5400.6 1621.13  5440.6 1613.86  5470.6 1611.56  5500.6 1615.01  5660.7 1614.08
  5710.7 1611.69  5878.1 1611.42  5950.9 1611.46  5958.4 1607.57  5958.9 1607.07
  5983.3 1607.57  6000.9 1614.75  6048.2 1623.52  6090.9 1631.94  6177.9 1633.19
#Mann=9,-1,0
  4434.8   0.035       0  4608.7    0.07       0  4944.8   0.035       0
  5004.9    0.07       0  5125.5   0.035       0  5878.1    0.07       0
  5958.4   0.035       0  5983.3    0.07       0  6048.2   0.035       0
Bank Sta=5958.4,5983.3
Exp/Cntr=0.3,0.1

Type RM Length L Ch R = 1,41785,698,698,698
BEGIN DESCRIPTION:
Mapping XS 54fd50cb
END DESCRIPTION:
XS GIS Cut Line= 3
      1675333.49      7000088.62      1676153.79      6999739.67
      1676980.38      6999503.13
#Sta/Elev= 30
  4110.5 1659.87  4114.1 1659.86  4232.1 1654.62  4303.0 1647.64  4340.3 1646.30
  4503.0 1622.94  4532.1 1623.60  4537.5 1625.39  4555.7 1625.84  4561.1 1627.96
  4600.0 1628.60  4637.5 1628.33  4761.1 1615.47  4837.5 1613.33  4948.9 1613.53
  5022.5 1607.20  5034.4 1608.29  5044.8 1613.64  5055.2 1615.15  5563.0 1612.27
  5609.7 1610.76  5646.0 1605.50  5646.5 1605.00  5670.9 1605.50  5689.7 1613.58
  5700.1 1616.87  5710.5 1617.54  5716.2 1620.88  5761.4 1627.94  5861.7 1631.40
#Mann=7,-1,0
  4110.5   0.035       0  4114.1    0.07       0  4600.0   0.035       0
  5563.0    0.07       0  5646.0   0.035       0  5670.9    0.07       0
  5761.4   0.035       0
Bank Sta=5646,5670.9
Exp/Cntr=0.3,0.1

Type RM Length L Ch R = 1,41087,882,882,882
BEGIN DESCRIPTION:
Mapping XS c229b531
END DESCRIPTION:
XS GIS Cut Line= 4
      1676050.08      7000637.47      1676452.87      7000047.17
      1676536.20      6999772.87      1676992.77      6999572.26
#Sta/Elev= 30
  4275.7 1630.72  4394.9 1627.93  4436.9 1624.94  4589.3 1619.39  4861.6 1614.26
  4876.5 1611.10  4893.5 1609.70  4927.4 1606.30  4963.3 1608.07  4999.3 1606.79
  5031.3 1609.03  5048.1 1612.15  5053.3 1610.76  5081.0 1612.28  5319.4 1611.68
  5457.9 1607.99  5494.1 1607.20  5500.0 1605.38  5516.0 1606.76  5537.8 1605.04
  5552.2 1605.47  5569.0 1603.43  5569.5 1602.93  5594.0 1603.43  5614.3 1608.43
  5636.1 1615.93  5651.0 1618.13  5674.4 1624.02  5713.0 1626.43  5775.7 1628.18
#Mann=7,-1,0
  4275.7   0.035       0  4893.5    0.07       0  4999.3   0.035       0
  5457.9    0.07       0  5569.0   0.035       0  5594.0    0.07       0
  5713.0   0.035       0
Bank Sta=5569,5594
Exp/Cntr=0.3,0.1

Type RM Length L Ch R = 1,40205,347,347,347
BEGIN DESCRIPTION:
Mapping XS 0e12c115
END DESCRIPTION:
XS GIS Cut Line= 3
      1676077.85      7000706.91      1677029.26      6999970.78
      1677764.53      6999412.40
#Sta/Elev= 30
  3790.9 1630.56  3988.3 1626.50  4079.8 1620.41  4123.2 1616.10  4251.8 1612.04
  4365.9 1610.33  4573.7 1611.37  4587.8 1611.28  4843.1 1610.61  4878.4 1609.59
  4899.9 1608.20  4928.2 1604.68  4950.5 1604.97  4966.4 1603.23  4973.5 1601.45
  4974.0 1600.95  4998.8 1601.45  5013.6 1602.18  5027.8 1606.00  5056.9 1611.40
  5077.8 1613.40  5185.9 1619.67  5313.3 1623.47  5377.8 1625.91  5400.1 1627.80
  5620.5 1635.55  5784.8 1645.87  5828.5 1647.24  5855.7 1649.51  5917.1 1653.28
#Mann=8,-1,0
  3790.9   0.035       0  4573.7    0.07       0  4587.8   0.035       0
  4966.4    0.07       0  4973.5    0.07       0  4998.8    0.07       0
  5313.3   0.035       0  5855.7    0.07       0
Bank Sta=4973.5,4998.8
Exp/Cntr=0.3,0.1

Type RM Length L Ch R = 1,39858,398,398,398
BEGIN DESCRIPTION:
Mapping XS bf263df4
END DESCRIPTION:
XS GIS Cut Line= 3
      1676202.89      7000849.24      1677244.54      7000234.67
      1677782.75      6999616.60
#Sta/Elev= 30
  3787.0 1626.15  3978.7 1624.72  4068.1 1620.31  4074.4 1617.77  4095.8 1615.42
  4132.9 1608.70  4170.0 1607.87  4607.1 1609.36  4724.2 1608.35  4745.6 1609.38
  4825.6 1608.69  4868.5 1604.98  4915.4 1602.50  4950.5 1604.02  4951.5 1600.40
  4952.0 1599.90  4976.8 1600.40  4979.8 1603.04  4996.4 1602.21  5008.3 1605.13
  5051.1 1609.62  5150.8 1613.12  5207.1 1617.49  5298.9 1620.99  5350.0 1624.77
  5533.4 1637.28  5589.4 1643.08  5632.1 1645.67  5791.7 1645.64  5816.0 1646.44
#Mann=7,-1,0
  3787.0   0.035       0  4868.5    0.07       0  4951.5    0.07       0
  4976.8    0.07       0  5207.1   0.035       0  5350.0    0.07       0
  5791.7   0.035       0
Bank Sta=4951.5,4976.8
Exp/Cntr=0.3,0.1

Type RM Length L Ch R = 1,39460,676,676,676
BEGIN DESCRIPTION:
Fish Creek 68.0
END DESCRIPTION:
XS GIS Cut Line= 3
      1676065.86      7000967.86      1677354.91      7000597.13
      1677929.99      6999713.01
#Sta/Elev= 30
  3658.7 1627.58  3666.8 1627.43  3771.0 1624.94  3853.7 1622.83  3897.9 1624.92
  3907.5 1623.73  4053.2 1623.22  4105.2 1620.83  4144.1 1616.14  4188.5 1606.99
  4230.1 1605.32  4907.2 1608.16  4942.7 1607.30  4948.1 1604.69  4956.2 1598.12
  4956.7 1597.62  4981.5 1598.12  5007.1 1598.53  5034.7 1603.80  5043.4 1603.19
  5070.5 1606.32  5152.1 1606.05  5187.8 1607.77  5291.0 1609.18  5360.3 1611.10
  5505.2 1621.10  5571.6 1624.04  5613.9 1628.22  5722.6 1635.37  6054.7 1652.44
#Mann=8,-1,0
  3658.7   0.035       0  3666.8    0.07       0  3771.0   0.035       0
  4907.2    0.07       0  4956.2    0.07       0  4981.5    0.07       0
  5187.8   0.035       0  5291.0    0.07       0
Bank Sta=4956.2,4981.5
Exp/Cntr=0.3,0.1

Type RM Length L Ch R = 1,38784,420,420,420
BEGIN DESCRIPTION:
Fish Creek 66.0
END DESCRIPTION:
XS GIS Cut Line= 3
      1676434.80      7000928.79      1677441.88      7001201.32
      1677854.08      7002560.70
#Sta/Elev= 30
  3956.7 1621.66  4166.8 1614.69  4201.4 1605.86  4236.1 1602.37  4551.1 1604.49
  4612.7 1604.77  4871.4 1603.63  4932.9 1603.33  4963.1 1598.98  4982.5 1597.33
  4999.0 1600.38  5016.1 1597.09  5042.8 1596.83  5043.3 1596.33  5073.6 1596.83
  5080.1 1603.91  5134.5 1606.07  5153.3 1602.95  5195.1 1603.43  5233.2 1609.63
  5362.3 1614.58  5506.9 1626.12  5540.5 1631.65  5641.8 1648.32  5763.0 1657.96
  5858.2 1661.64  5927.8 1662.85  6188.2 1667.95  6260.4 1667.96  6420.5 1666.30
#Mann=15,-1,0
  3956.7   0.035       0  4551.1    0.07       0  4612.7   0.035       0
  4871.4    0.07       0  4963.1   0.035       0  5016.1    0.07       0
  5042.8   0.035       0  5073.6    0.07       0  5540.5   0.035       0
  5641.8    0.07       0  5763.0   0.035       0  5858.2    0.07       0
  5927.8   0.035       0  6188.2    0.07       0  6260.4   0.035       0
Bank Sta=5042.8,5073.6
Exp/Cntr=0.3,0.1

Type RM Length L Ch R = 1,38364,1096,1096,1096
BEGIN DESCRIPTION:
Mapping XS e1c27b4f
END DESCRIPTION:
XS GIS Cut Line= 3
      1676105.00      7001098.08      1677159.65      7001484.35
      1677537.24      7002369.74
#Sta/Elev= 30
  3877.9 1625.41  4121.3 1614.76  4250.6 1608.57  4304.2 1602.66  4346.5 1604.63
  4440.9 1602.48  4471.4 1599.97  4484.9 1596.53  4501.9 1600.18  4527.1 1600.51
  4593.4 1596.56  4769.8 1599.75  4850.8 1601.85  4938.3 1601.73  4978.5 1595.73
  4979.0 1595.23  5009.4 1595.73  5026.5 1600.88  5039.6 1604.37  5194.8 1607.60
  5374.7 1614.27  5418.1 1617.99  5440.3 1623.26  5510.6 1630.75  5535.7 1635.61
  5634.7 1646.73  5669.2 1653.35  5722.5 1658.54  5812.1 1658.16  5963.6 1656.65
#Mann=13,-1,0
  3877.9   0.035       0  4121.3    0.07       0  4440.9   0.035       0
  4769.8    0.07       0  4850.8   0.035       0  4978.5   0.035       0
  5009.4   0.035       0  5026.5    0.07       0  5039.6   0.035       0
  5194.8    0.07       0  5510.6   0.035       0  5535.7    0.07       0
  5812.1   0.035       0
Bank Sta=4978.5,5009.4
Exp/Cntr=0.3,0.1

Type RM Length L Ch R = 1,37268,461,461,461
BEGIN DESCRIPTION:
Mapping XS be6adde7
END DESCRIPTION:
XS GIS Cut Line= 3
      1675631.89      7001154.50      1676313.29      7001536.43
      1677328.92      7002261.26
#Sta/Elev= 30
  4223.8 1637.03  4410.8 1632.17  4721.2 1628.17  4743.2 1627.68  4794.1 1624.28
  4815.8 1621.96  4846.4 1615.68  4891.1 1610.89  4918.5 1603.27  4946.4 1591.08
  4946.9 1590.58  4977.4 1591.08  4977.9 1591.93  4984.0 1593.26  4999.6 1595.76
  5020.9 1595.63  5071.3 1598.71  5192.9 1599.28  5225.4 1600.44  5297.6 1600.98
  5343.6 1601.59  5637.9 1602.26  5822.9 1607.83  5961.1 1613.87  6011.5 1620.79
  6068.0 1624.55  6097.5 1629.20  6118.4 1631.26  6133.2 1635.08  6252.7 1644.38
#Mann=8,-1,0
  4223.8   0.035       0  4721.2    0.07       0  4946.4    0.07       0
  4977.4    0.07       0  5225.4   0.035       0  5297.6    0.07       0
  5343.6   0.035       0  5822.9    0.07       0
Bank Sta=4946.4,4977.4
Exp/Cntr=0.3,0.1
