HEC-RAS study Fish Creek.prj: Fish Creek Base Level Engineering

--- Fish Creek.g01 (geometry) --- (continued)

Type RM Length L Ch R = 1,36807,375,375,375
BEGIN DESCRIPTION:
Mapping XS 2d889602
END DESCRIPTION:
XS GIS Cut Line= 3
      1675214.37      7001360.24      1676058.08      7001896.67
      1677667.49      7002667.52
#Sta/Elev= 30
  4010.8 1649.23  4062.9 1647.16  4197.5 1638.98  4313.9 1629.68  4501.9 1623.38
  4559.5 1618.83  4595.9 1613.05  4632.3 1613.53  4684.0 1619.45  4689.9 1617.39
  4714.2 1617.47  4762.8 1615.71  4835.6 1617.15  4887.2 1613.53  4929.6 1604.42
  4965.7 1589.19  4966.2 1588.69  4996.7 1589.19  5007.6 1589.95  5030.1 1595.86
  5069.9 1597.80  5324.7 1598.95  5375.6 1597.21  5512.8 1600.37  5639.9 1602.91
  5933.9 1609.44  6315.6 1625.61  6417.6 1634.28  6548.0 1650.10  6795.1 1656.22
#Mann=10,-1,0
  4010.8   0.035       0  4062.9    0.07       0  4197.5   0.035       0
  4714.2    0.07       0  4965.7    0.07       0  4996.7    0.07       0
  5007.6   0.035       0  5512.8    0.07       0  5639.9   0.035       0
  5933.9    0.07       0
Bank Sta=4965.7,4996.7
Exp/Cntr=0.3,0.1

Type RM Length L Ch R = 1,36432,544,544,544
BEGIN DESCRIPTION:
Mapping XS 12a6a9c5
END DESCRIPTION:
XS GIS Cut Line= 3
      1674917.49      7001438.37      1675854.96      7002198.76
      1676979.95      7003177.91
#Sta/Elev= 30
  3802.7 1655.91  3976.1 1650.60  4110.9 1645.08  4120.3 1644.37  4286.5 1634.45
  4308.0 1633.20  4348.3 1629.41  4400.4 1627.59  4609.8 1625.19  4696.7 1621.26
  4767.1 1604.25  4795.8 1599.02  4815.4 1597.68  4881.1 1597.34  4920.5 1593.72
  5015.1 1590.62  5015.6 1590.12  5046.1 1590.62  5059.1 1594.61  5078.0 1596.77
  5406.6 1595.40  5661.0 1603.15  5841.0 1612.07  5895.6 1615.21  5965.8 1622.46
  6114.9 1647.32  6328.9 1657.00  6443.5 1658.06  6470.2 1658.20  6501.2 1658.36
#Mann=17,-1,0
  3802.7   0.035       0  3976.1    0.07       0  4110.9   0.035       0
  4120.3    0.07       0  4286.5   0.035       0  4308.0    0.07       0
  4400.4   0.035       0  4609.8    0.07       0  4815.4   0.035       0
  4920.5    0.07       0  5015.1    0.07       0  5046.1    0.07       0
  5078.0   0.035       0  5841.0    0.07       0  6328.9   0.035       0
  6443.5    0.07       0  6470.2   0.035       0
Bank Sta=5015.1,5046.1
Exp/Cntr=0.3,0.1

Type RM Length L Ch R = 1,35888,918,918,918
BEGIN DESCRIPTION:
Mapping XS eb1fadea
END DESCRIPTION:
XS GIS Cut Line= 3
      1674714.33      7001922.71      1675594.54      7002646.67
      1676764.89      7003484.13
#Sta/Elev= 30
  3859.0 1652.27  4081.4 1648.74  4175.7 1645.10  4303.4 1636.84  4389.5 1624.97
  4453.3 1619.58  4523.7 1596.27  4552.3 1593.30  4585.9 1592.96  4729.6 1597.06
  4831.8 1595.58  4929.0 1592.72  4948.7 1589.31  4949.2 1588.81  4979.7 1589.31
  4995.8 1592.49  5028.4 1589.58  5078.7 1590.27  5114.4 1594.20  5153.6 1594.76
  5200.4 1598.43  5301.1 1598.47  5393.2 1603.99  5872.8 1617.56  6161.1 1631.04
  6204.3 1634.88  6282.7 1645.29  6347.8 1648.18  6394.3 1652.57  6437.8 1655.06
#Mann=9,-1,0
  3859.0   0.035       0  4081.4    0.07       0  4585.9   0.035       0
  4831.8    0.07       0  4948.7    0.07       0  4979.7    0.07       0
  5153.6   0.035       0  5872.8    0.07       0  6394.3   0.035       0
Bank Sta=4948.7,4979.7
Exp/Cntr=0.3,0.1

Type RM Length L Ch R = 1,34970,410,410,410
BEGIN DESCRIPTION:
Mapping XS b74b196f
END DESCRIPTION:
XS GIS Cut Line= 3
      1674609.39      7002421.28      1674835.27      7002708.50
      1675491.11      7003479.89
#Sta/Elev= 30
  4634.6 1645.26  4700.3 1643.44  4721.2 1641.55  4757.6 1635.35  4785.3 1632.89
  4793.4 1630.05  4814.2 1626.54  4892.8 1606.80  4913.6 1602.78  4928.1 1598.19
  4935.8 1593.45  4942.5 1587.85  4947.7 1581.80  4948.2 1581.30  4979.0 1581.80
  4985.9 1583.01  5003.0 1583.40  5006.6 1587.29  5013.2 1589.61  5035.2 1591.91
  5120.3 1590.90  5134.0 1590.04  5148.3 1591.51  5191.1 1590.76  5326.2 1594.24
  5574.4 1595.81  5603.0 1596.47  5609.5 1597.62  5681.0 1597.87  6012.5 1604.35
#Mann=4,-1,0
  4634.6    0.07       0  4947.7    0.07       0  4979.0    0.07       0
  5120.3   0.035       0
Bank Sta=4947.7,4979
Exp/Cntr=0.3,0.1

Type RM Length L Ch R = 1,34560,440,440,440
BEGIN DESCRIPTION:
Mapping XS c649f305
END DESCRIPTION:
XS GIS Cut Line= 3
      1674242.41      7002677.60      1674511.05      7002929.84
      1675067.12      7003518.67
#Sta/Elev= 30
  4631.5 1628.08  4640.7 1627.09  4683.1 1627.74  4718.3 1625.56  4725.6 1626.12
  4768.1 1622.10  4775.0 1620.22  4791.1 1618.49  4796.4 1618.11  4845.8 1606.83
  4930.8 1590.72  4937.6 1588.00  4959.1 1584.69  4973.3 1584.20  5002.2 1586.43
  5017.5 1589.77  5065.3 1591.52  5121.6 1590.56  5149.9 1588.07  5185.5 1586.99
  5205.0 1582.89  5205.5 1582.39  5236.3 1582.89  5242.1 1588.37  5263.2 1593.12
  5284.6 1591.40  5324.2 1591.41  5652.3 1592.60  5772.5 1594.39  5809.9 1593.85
#Mann=6,-1,0
  4631.5   0.035       0  4791.1    0.07       0  5017.5   0.035       0
  5205.0    0.07       0  5236.3   0.035       0  5324.2   0.035       0
Bank Sta=5205,5236.3
Exp/Cntr=0.3,0.1

Type RM Length L Ch R = 1,34120,474,474,474
BEGIN DESCRIPTION:
Mapping XS ca40fabc
END DESCRIPTION:
XS GIS Cut Line= 3
      1674024.50      7002921.41      1674304.92      7003267.97
      1675900.14      7004162.88
#Sta/Elev= 30
  4554.2 1614.70  4637.9 1616.61  4693.9 1614.28  4772.3 1592.45  4786.7 1589.77
  4819.4 1588.31  4984.9 1586.28  4996.8 1584.28  4998.1 1579.29  4998.6 1578.79
  5029.4 1579.29  5029.7 1581.07  5051.4 1582.80  5089.1 1580.37  5110.8 1584.20
  5116.5 1586.84  5132.4 1587.53  5148.4 1590.69  5231.9 1591.17  5699.5 1590.17
  5770.3 1593.85  6110.3 1601.03  6394.6 1609.96  6513.3 1613.99  6517.7 1614.11
  6580.4 1616.91  6642.1 1622.45  6720.0 1629.58  6791.5 1641.49  6829.1 1642.78
#Mann=10,-1,0
  4554.2    0.07       0  4819.4   0.035       0  4984.9    0.07       0
  4998.1    0.07       0  5029.4    0.07       0  5231.9   0.035       0
  6394.6    0.07       0  6513.3   0.035       0  6517.7    0.07       0
  6642.1   0.035       0
Bank Sta=4998.1,5029.4
Exp/Cntr=0.3,0.1

Type RM Length L Ch R = 1,33646,1369,1369,1369
BEGIN DESCRIPTION:
Mapping XS 2769dc22
END DESCRIPTION:
XS GIS Cut Line= 3
      1673816.64      7003387.14      1674104.69      7003667.70
      1675609.65      7004223.15
#Sta/Elev= 30
  4597.9 1598.27  4719.1 1599.08  4762.4 1599.30  4868.1 1605.15  4887.4 1606.81
  4901.5 1605.56  4924.7 1596.89  4929.8 1593.27  4936.8 1591.71  4943.9 1587.21
  4950.9 1585.67  4958.1 1580.17  4977.7 1574.13  4978.2 1573.63  5009.0 1574.13
  5010.5 1576.98  5015.8 1578.35  5021.7 1582.51  5040.9 1586.46  5170.9 1585.91
  5395.4 1588.08  5481.4 1586.41  5592.4 1586.62  5825.2 1595.48  6022.2 1597.69
  6186.6 1601.43  6315.9 1605.03  6450.0 1610.77  6493.1 1613.48  6604.2 1624.93
#Mann=8,-1,0
  4597.9    0.07       0  4719.1   0.035       0  4762.4    0.07       0
  4868.1   0.035       0  4924.7    0.07       0  4977.7   0.035       0
  5009.0    0.07       0  6186.6    0.07       0
Bank Sta=4977.7,5009
Exp/Cntr=0.3,0.1

Type RM Length L Ch R = 1,32277,526,526,526
BEGIN DESCRIPTION:
Mapping XS 83bd36e2
END DESCRIPTION:
XS GIS Cut Line= 3
      1673151.46      7002999.32      1674019.53      7004774.52
      1674240.44      7005160.03
#Sta/Elev= 30
  3024.7 1626.24  3160.2 1622.85  3199.6 1619.05  3385.3 1613.07  3452.9 1611.89
  3538.5 1612.82  3661.0 1610.65  3735.7 1599.73  3801.9 1595.64  3880.4 1593.65
  4161.9 1590.44  4381.3 1585.38  4817.5 1583.34  4826.0 1583.17  4902.7 1580.91
  4961.0 1578.05  4971.3 1575.80  4978.0 1575.90  4983.4 1570.53  4984.0 1570.03
  5016.5 1570.53  5022.0 1576.58  5027.8 1579.88  5037.8 1584.83  5059.4 1592.32
  5177.3 1621.18  5198.9 1624.98  5290.3 1632.63  5338.5 1636.19  5445.1 1639.03
#Mann=9,-1,0
  3024.7   0.035       0  3538.5    0.07       0  3801.9   0.035       0
  4817.5    0.07       0  4826.0   0.035       0  4902.7    0.07       0
  4983.4    0.07       0  5016.5    0.07       0  5290.3   0.035       0
Bank Sta=4983.4,5016.5
Exp/Cntr=0.3,0.1

Type RM Length L Ch R = 1,31751,996,996,996
BEGIN DESCRIPTION:
Mapping XS 43e869a9
END DESCRIPTION:
XS GIS Cut Line= 3
      1672664.49      7003325.74      1673549.91      7004945.53
      1673987.33      7005513.14
#Sta/Elev= 30
  3164.1 1626.40  3391.7 1611.20  3418.3 1609.81  3510.5 1607.33  3658.8 1605.37
  3734.7 1596.55  3805.8 1593.58  4834.8 1580.51  4927.2 1578.26  4948.6 1568.98
  4949.2 1568.48  4981.7 1568.98  5001.5 1571.61  5008.7 1575.79  5043.9 1578.22
  5072.9 1590.12  5087.4 1594.61  5093.7 1594.68  5108.2 1604.37  5114.5 1604.87
  5122.7 1609.32  5129.0 1609.71  5137.2 1614.29  5143.5 1614.63  5164.7 1622.62
  5257.7 1632.29  5355.1 1635.65  5529.5 1642.02  5694.2 1644.63  5726.7 1645.04
#Mann=9,-1,0
  3164.1    0.07       0  3391.7   0.035       0  3418.3    0.07       0
  3510.5   0.035       0  4834.8    0.07       0  4948.6    0.07       0
  4981.7    0.07       0  5355.1   0.035       0  5694.2    0.07       0
Bank Sta=4948.6,4981.7
Exp/Cntr=0.3,0.1

Type RM Length L Ch R = 1,30755,655,655,655
BEGIN DESCRIPTION:
Mapping XS 6f9510b4
END DESCRIPTION:
XS GIS Cut Line= 3
      1671792.52      7003591.77      1672599.82      7004899.09
      1673563.38      7005711.60
#Sta/Elev= 30
  3466.4 1637.43  3792.1 1623.62  3843.8 1620.73  3901.0 1614.88  3959.0 1612.84
  4099.2 1598.25  4366.9 1586.01  4569.1 1579.70  4605.7 1582.01  4932.0 1577.62
  4947.4 1576.80  4984.1 1569.57  5018.0 1568.41  5018.6 1567.91  5051.3 1568.41
  5062.0 1571.74  5090.6 1574.07  5147.8 1572.74  5168.8 1576.12  5211.5 1575.61
  5225.8 1573.32  5240.1 1576.96  5361.0 1578.41  5694.0 1618.64  5765.4 1621.97
  5843.5 1629.02  5919.5 1630.93  6206.4 1631.62  6258.3 1631.83  6263.3 1632.06
#Mann=10,-1,0
  3466.4    0.07       0  3792.1   0.035       0  3843.8    0.07       0
  4099.2   0.035       0  5018.0   0.035       0  5051.3   0.035       0
  5168.8    0.07       0  5919.5   0.035       0  6206.4    0.07       0
  6258.3   0.035       0
Bank Sta=5018,5051.3
Exp/Cntr=0.3,0.1

Type RM Length L Ch R = 1,30100,409,409,409
BEGIN DESCRIPTION:
Mapping XS 1c7cfc6a
END DESCRIPTION:
XS GIS Cut Line= 3
      1670743.93      7004029.30      1672014.75      7005091.80
      1673465.00      7005903.66
#Sta/Elev= 30
  3353.4 1717.08  3530.7 1708.90  3672.6 1697.77  3862.4 1659.55  3976.4 1640.17
  4319.3 1604.10  4527.3 1592.70  4800.4 1578.79  4845.8 1578.05  4943.9 1575.19
  4950.5 1572.65  4954.6 1562.81  4955.2 1562.31  4988.0 1562.81  4993.4 1567.09
  5015.1 1568.07  5022.8 1567.87  5051.8 1567.51  5138.6 1575.62  5419.4 1576.39
  5668.3 1583.01  5728.8 1587.76  5808.7 1596.24  5920.0 1597.44  5996.8 1600.56
  6198.0 1611.10  6300.7 1614.05  6344.1 1611.91  6403.5 1617.81  6671.9 1631.28
#Mann=13,-1,0
  3353.4    0.07       0  3862.4   0.035       0  3976.4    0.07       0
  4527.3   0.035       0  4800.4    0.07       0  4845.8   0.035       0
  4954.6   0.035       0  4988.0   0.035       0  5015.1    0.07       0
  5022.8   0.035       0  5728.8    0.07       0  5920.0   0.035       0
  5996.8    0.07       0
Bank Sta=4954.6,4988
Exp/Cntr=0.3,0.1

Type RM Length L Ch R = 1,29691,722,722,722
BEGIN DESCRIPTION:
Mapping XS e802db09
END DESCRIPTION:
XS GIS Cut Line= 3
      1670841.10      7005077.90      1671855.03      7005439.02
      1673118.94      7005945.97
#Sta/Elev= 30
  3928.1 1708.44  3976.6 1703.78  4023.8 1695.78  4063.7 1685.42  4089.2 1675.07
  4143.5 1664.04  4344.0 1624.06  4489.2 1601.15  4541.0 1594.60  4590.4 1584.53
  4688.0 1578.42  4751.5 1575.01  4864.2 1573.80  4961.9 1566.63  4970.7 1561.54
  4971.3 1561.04  5004.2 1561.54  5017.8 1561.81  5036.6 1568.12  5079.8 1572.89
  5307.1 1575.23  5580.0 1580.24  5633.8 1585.33  5672.4 1593.49  5717.2 1598.72
  5812.9 1606.55  5902.8 1613.19  6023.7 1615.38  6149.6 1617.23  6366.2 1625.12
#Mann=12,-1,0
  3928.1    0.07       0  4023.8   0.035       0  4143.5    0.07       0
  4344.0   0.035       0  4489.2    0.07       0  4688.0   0.035       0
  4970.7   0.035       0  5004.2   0.035       0  5307.1    0.07       0
  5812.9   0.035       0  6023.7    0.07       0  6149.6   0.035       0
Bank Sta=4970.7,5004.2
Exp/Cntr=0.3,0.1

Type RM Length L Ch R = 1,28969,497,497,497
BEGIN DESCRIPTION:
Mapping XS e4935a84
END DESCRIPTION:
XS GIS Cut Line= 3
      1670889.79      7005902.42      1671405.38      7005988.35
      1673124.13      7006092.52
#Sta/Elev= 30
  4473.7 1642.49  4597.2 1623.04  4773.0 1607.25  4793.3 1603.45  4864.2 1596.80
  4894.6 1593.48  4935.2 1582.49  4962.2 1568.44  4975.7 1563.55  4976.9 1558.17
  4977.5 1557.67  5010.5 1558.17  5016.1 1561.86  5036.1 1562.22  5072.2 1568.69
  5106.2 1570.39  5176.3 1569.11  5436.8 1574.15  5729.8 1576.37  5937.7 1582.22
  5967.8 1584.73  6064.0 1600.28  6188.2 1601.09  6218.3 1603.74  6268.3 1612.80
  6365.4 1618.37  6448.7 1624.12  6590.9 1628.16  6635.3 1628.86  6718.3 1630.13
#Mann=8,-1,0
  4473.7    0.07       0  4864.2   0.035       0  4976.9   0.035       0
  5010.5   0.035       0  5729.8    0.07       0  6365.4   0.035       0
  6590.9    0.07       0  6635.3   0.035       0
Bank Sta=4976.9,5010.5
Exp/Cntr=0.3,0.1

Type RM Length L Ch R = 1,28472,463,463,463
BEGIN DESCRIPTION:
Mapping XS 9b8ea2b0
END DESCRIPTION:
XS GIS Cut Line= 3
      1670918.41      7006519.60      1671397.57      7006485.75
      1672808.99      7006410.23
#Sta/Elev= 30
  4512.3 1611.02  4663.5 1602.73  4699.4 1601.12  4719.4 1597.52  4739.5 1596.22
  4819.7 1596.19  4849.7 1590.82  4929.9 1586.18  4988.9 1562.30  4992.7 1562.30
  4993.3 1555.38  4993.9 1554.88  5026.9 1555.38  5030.1 1560.13  5050.2 1559.50
  5080.2 1563.25  5150.3 1567.45  5249.9 1567.56  5310.5 1570.73  5440.2 1572.25
  5795.3 1575.12  5921.4 1577.27  6001.5 1581.56  6051.6 1588.17  6091.7 1596.69
  6151.7 1605.10  6166.9 1609.12  6211.8 1612.77  6271.9 1620.81  6406.1 1625.10
#Mann=7,-1,0
  4512.3   0.035       0  4663.5    0.07       0  4993.3   0.035       0
  5026.9    0.07       0  5249.9    0.07       0  5440.2   0.035       0
  5795.3    0.07       0
Bank Sta=4993.3,5026.9
Exp/Cntr=0.3,0.1

Type RM Length L Ch R = 1,28009,295,295,295
BEGIN DESCRIPTION:
Mapping XS e920bb29
END DESCRIPTION:
XS GIS Cut Line= 3
      1670892.39      7007084.70      1671504.34      7006899.81
      1672961.37      7006525.15
#Sta/Elev= 30
  4360.0 1597.80  4563.0 1596.48  4582.5 1596.19  4664.2 1594.91  4786.6 1591.71
  4864.2 1587.96  4895.5 1584.24  4920.4 1575.42  4926.8 1571.21  4953.3 1560.58
  4979.1 1554.14  4988.6 1554.48  4993.4 1553.97  4994.1 1553.47  5027.1 1553.97
  5031.4 1559.82  5050.8 1560.53  5072.2 1564.93  5092.9 1566.76  5247.8 1566.47
  5352.0 1569.90  5774.3 1574.44  5852.6 1576.53  5960.2 1580.06  6011.8 1584.51
  6135.7 1603.74  6166.7 1609.91  6239.0 1619.65  6268.1 1622.02  6503.7 1626.93
#Mann=10,-1,0
  4360.0   0.035       0  4563.0    0.07       0  4582.5   0.035       0
  4664.2    0.07       0  4786.6   0.035       0  4988.6    0.07       0
  4993.4    0.07       0  5027.1    0.07       0  5050.8   0.035       0
  5852.6    0.07       0
Bank Sta=4993.4,5027.1
Exp/Cntr=0.3,0.1

Type RM Length L Ch R = 1,27714,322,322,322
BEGIN DESCRIPTION:
Mapping XS 45f3f76a
END DESCRIPTION:
XS GIS Cut Line= 3
      1670967.92      7007355.53      1671556.42      7007178.46
      1673224.78      7006652.71
#Sta/Elev= 30
  4385.3 1591.50  4634.0 1594.61  4780.1 1590.10  4840.9 1589.89  4862.6 1587.67
  4873.1 1586.36  4904.4 1575.32  4912.2 1571.04  4948.9 1561.53  4967.1 1557.50
  4983.4 1557.69  4999.1 1554.98  4999.8 1554.48  5033.0 1554.98  5061.3 1561.78
  5166.1 1566.02  5549.6 1573.38  5684.3 1573.07  5927.2 1577.65  6045.5 1582.09
  6109.8 1588.67  6153.1 1597.53  6244.9 1605.24  6250.2 1607.05  6277.3 1607.95
  6282.5 1609.73  6347.3 1612.15  6424.3 1619.65  6551.9 1623.67  6749.1 1622.87
#Mann=6,-1,0
  4385.3   0.035       0  4634.0    0.07       0  4948.9   0.035       0
  4999.1   0.035       0  5033.0   0.035       0  5927.2    0.07       0
Bank Sta=4999.1,5033
Exp/Cntr=0.3,0.1

Type RM Length L Ch R = 1,27392,303,303,303
BEGIN DESCRIPTION:
Mapping XS 84430e10
END DESCRIPTION:
XS GIS Cut Line= 3
      1671137.98      7007470.12      1671606.77      7007485.32
      1672986.95      7007652.41
#Sta/Elev= 30
  4533.1 1593.47  4689.9 1595.03  4820.3 1593.96  4850.3 1591.56  4880.3 1584.66
  4928.0 1570.26  4933.0 1570.98  4940.3 1567.75  4970.4 1559.23  4973.4 1553.76
  4974.1 1553.26  5007.3 1553.76  5028.6 1555.14  5050.7 1558.53  5071.0 1559.12
  5101.1 1562.51  5229.7 1565.24  5614.8 1566.77  5835.7 1576.40  5917.0 1581.00
  5967.4 1588.40  5981.9 1589.05  5987.5 1591.16  6037.9 1598.36  6063.8 1603.81
  6158.8 1608.23  6219.2 1613.34  6269.6 1616.00  6353.6 1618.58  6392.4 1619.67
#Mann=7,-1,0
  4533.1   0.035       0  4689.9    0.07       0  4973.4    0.07       0
  5007.3    0.07       0  5028.6   0.035       0  5835.7    0.07       0
  6353.6   0.035       0
Bank Sta=4973.4,5007.3
Exp/Cntr=0.3,0.1

Type RM Length L Ch R = 1,27089,814,814,814
BEGIN DESCRIPTION:
Mapping XS 67a5f7d0
END DESCRIPTION:
XS GIS Cut Line= 3
      1671178.38      7007622.03      1671652.34      7007770.47
      1672537.78      7008275.69
#Sta/Elev= 30
  4500.6 1592.77  4512.3 1592.72  4632.9 1593.56  4696.2 1590.50  4767.9 1584.51
  4821.9 1573.25  4870.5 1566.34  4946.6 1561.71  4967.8 1558.42  5004.2 1557.19
  5014.8 1554.89  5017.9 1554.40  5018.6 1553.90  5051.9 1554.40  5084.9 1555.81
  5115.5 1559.00  5249.1 1562.34  5283.6 1564.15  5355.0 1563.53  5432.6 1562.63
  5509.7 1560.12  5547.2 1561.21  5576.0 1566.53  5599.0 1569.02  5627.8 1575.77
  5702.6 1588.39  5745.9 1598.11  5817.8 1609.83  5848.2 1613.10  6016.7 1621.67
#Mann=10,-1,0
  4500.6   0.035       0  4512.3    0.07       0  4946.6   0.035       0
  5014.8    0.07       0  5017.9   0.035       0  5051.9    0.07       0
  5115.5   0.035       0  5249.1    0.07       0  5355.0   0.035       0
  5432.6    0.07       0
Bank Sta=5017.9,5051.9
Exp/Cntr=0.3,0.1

Type RM Length L Ch R = 1,26275,786,786,786
BEGIN DESCRIPTION:
Mapping XS 62a62988
END DESCRIPTION:
XS GIS Cut Line= 3
      1671223.93      7007712.85      1671757.81      7008489.80
      1672259.21      7008943.65
#Sta/Elev= 30
  4060.6 1591.60  4137.8 1585.63  4158.7 1582.62  4188.2 1582.05  4225.5 1578.58
  4309.5 1568.58  4373.9 1564.65  4430.8 1562.87  4836.4 1559.73  4884.7 1559.75
  4928.3 1557.71  4956.4 1553.25  4986.2 1553.02  4990.2 1548.33  4990.8 1547.83
  5024.2 1548.33  5042.3 1552.56  5063.9 1564.04  5078.1 1567.14  5127.5 1573.26
  5170.0 1585.16  5198.4 1590.25  5269.3 1598.52  5304.5 1603.90  5339.7 1605.22
  5347.1 1606.61  5410.7 1606.73  5424.8 1608.01  5516.8 1607.16  5679.6 1609.75
#Mann=5,-1,0
  4060.6    0.07       0  4225.5   0.035       0  4836.4    0.07       0
  4990.2    0.07       0  5024.2    0.07       0
Bank Sta=4990.2,5024.2
Exp/Cntr=0.3,0.1

Type RM Length L Ch R = 1,25489,845,845,845
BEGIN DESCRIPTION:
Mapping XS 074775d8
END DESCRIPTION:
XS GIS Cut Line= 3
      1671067.70      7007719.40      1671213.10      7008893.45
      1671369.35      7009611.73
#Sta/Elev= 30
  3822.4 1590.34  4022.5 1580.35  4123.3 1568.79  4203.8 1564.57  4653.5 1559.98
  4727.9 1556.33  4894.9 1555.57  4949.5 1555.25  4969.7 1552.49  4977.4 1549.74
  4982.5 1550.52  4987.7 1548.10  4988.5 1547.60  5022.6 1548.10  5030.5 1548.26
  5036.8 1552.17  5094.7 1556.67  5153.3 1558.90  5179.0 1562.86  5195.5 1562.82
  5255.7 1563.81  5272.1 1567.77  5321.2 1573.97  5409.2 1589.12  5414.3 1588.53
  5463.5 1594.61  5507.4 1601.30  5583.2 1605.55  5706.0 1604.78  5740.5 1606.24
#Mann=8,-1,0
  3822.4    0.07       0  4203.8   0.035       0  4894.9    0.07       0
  4987.7    0.07       0  5022.6    0.07       0  5094.7   0.035       0
  5195.5    0.07       0  5463.5   0.035       0
Bank Sta=4987.7,5022.6
Exp/Cntr=0.3,0.1

Type RM Length L Ch R = 1,24644,645,645,645
BEGIN DESCRIPTION:
Mapping XS 5ac945de
END DESCRIPTION:
XS GIS Cut Line= 3
      1669838.96      7007786.23      1670461.37      7008645.62
      1671216.57      7009669.04
#Sta/Elev= 30
  3944.6 1602.21  4014.6 1600.17  4131.4 1590.81  4201.0 1585.68  4443.8 1577.68
  4525.8 1568.69  4573.7 1563.61  4749.2 1559.99  4873.0 1559.06  4931.8 1555.84
  4946.5 1553.54  4964.4 1546.02  4965.2 1545.52  4999.6 1546.02  5002.9 1548.28
  5045.9 1546.59  5146.7 1553.32  5259.4 1553.87  5375.4 1555.30  5489.5 1553.32
  5528.4 1555.52  5567.9 1554.37  5589.7 1550.81  5610.6 1551.78  5639.8 1561.12
  5725.4 1579.36  5804.0 1591.35  5874.6 1597.81  6025.3 1602.55  6277.6 1604.58
#Mann=12,-1,0
  3944.6   0.035       0  4131.4    0.07       0  4525.8   0.035       0
  4749.2    0.07       0  4964.4    0.07       0  4999.6    0.07       0
  5146.7   0.035       0  5259.4    0.07       0  5375.4   0.035       0
  5528.4    0.07       0  5874.6   0.035       0  6025.3    0.07       0
Bank Sta=4964.4,4999.6
Exp/Cntr=0.3,0.1

Type RM Length L Ch R = 1,23999,1095,1095,1095
BEGIN DESCRIPTION:
Mapping XS bf857fb9
END DESCRIPTION:
XS GIS Cut Line= 3
      1669471.79      7008119.58      1670240.01      7009210.72
      1670910.94      7010029.88
#Sta/Elev= 30
  3670.3 1610.77  3851.8 1598.36  3944.3 1589.59  4066.3 1564.47  4108.6 1559.94
  4175.9 1557.12  4211.3 1556.11  4283.8 1554.72  4563.8 1551.84  4641.5 1551.95
  4681.4 1551.87  4955.6 1547.83  4977.0 1542.83  5000.0 1544.16  5023.8 1540.48
  5024.5 1539.98  5059.0 1540.48  5063.6 1546.84  5084.4 1544.61  5169.3 1557.52
  5245.6 1562.94  5250.3 1563.27  5426.1 1574.48  5475.6 1574.99  5496.4 1572.46
  5525.1 1575.43  5565.6 1574.58  5702.4 1591.70  5815.8 1600.81  6063.6 1607.47
#Mann=12,-1,0
  3670.3    0.07       0  4175.9   0.035       0  4211.3    0.07       0
  4283.8   0.035       0  4563.8    0.07       0  4641.5   0.035       0
  4681.4    0.07       0  5023.8    0.07       0  5059.0    0.07       0
  5245.6   0.035       0  5250.3    0.07       0  5565.6   0.035       0
Bank Sta=5023.8,5059
Exp/Cntr=0.3,0.1

Type RM Length L Ch R = 1,22904,689,689,689
BEGIN DESCRIPTION:
Mapping XS dc4c9712
END DESCRIPTION:
XS GIS Cut Line= 4
      1669084.56      7008234.37      1669355.38      7008852.39
      1669660.93      7009453.08      1670410.50      7010258.17
#Sta/Elev= 30
  4334.4 1635.31  4497.1 1608.18  4633.2 1596.92  4665.9 1596.08  4747.2 1587.48
  4822.8 1568.63  4846.2 1560.00  4892.9 1549.43  4950.6 1546.94  4991.0 1540.67
  5004.0 1538.09  5009.0 1533.66  5009.8 1533.16  5044.3 1533.66  5049.1 1540.77
  5059.1 1542.03  5094.0 1542.68  5138.9 1539.31  5175.9 1542.77  5192.6 1547.04
  5237.1 1549.04  5609.7 1552.66  6017.9 1561.27  6064.4 1564.75  6184.6 1585.50
  6269.6 1593.91  6361.5 1598.57  6485.4 1601.12  6652.9 1605.35  6783.1 1606.43
#Mann=7,-1,0
  4334.4    0.07       0  4991.0   0.035       0  5009.0   0.035       0
  5044.3   0.035       0  6017.9    0.07       0  6485.4   0.035       0
  6652.9    0.07       0
Bank Sta=5009,5044.3
Exp/Cntr=0.3,0.1

Type RM Length L Ch R = 1,22215,831,831,831
BEGIN DESCRIPTION:
Mapping XS 18eaea9b
END DESCRIPTION:
XS GIS Cut Line= 3
      1668657.48      7008487.85      1669032.46      7009369.75
      1669532.38      7010543.18
#Sta/Elev= 30
  4048.7 1615.42  4154.7 1603.02  4505.5 1577.89  4723.4 1570.81  4842.0 1569.44
  4871.1 1564.64  4876.5 1559.02  4900.2 1551.54  4923.8 1548.48  4929.3 1543.84
  4952.9 1538.13  4994.2 1534.16  5100.1 1533.70  5105.6 1533.41  5106.1 1530.97
  5106.9 1530.47  5141.5 1530.97  5146.4 1534.72  5186.3 1538.16  5205.5 1542.46
  5229.1 1541.01  5252.8 1544.21  5481.7 1546.40  5689.8 1553.90  5763.3 1561.17
  5768.8 1564.64  5792.4 1564.33  5892.4 1582.54  5996.3 1594.29  6282.5 1606.14
#Mann=8,-1,0
  4048.7    0.07       0  4505.5   0.035       0  4723.4    0.07       0
  5106.1    0.07       0  5141.5    0.07       0  5186.3   0.035       0
  5689.8    0.07       0  5996.3   0.035       0
Bank Sta=5106.1,5141.5
Exp/Cntr=0.3,0.1

Type RM Length L Ch R = 1,21384,779,779,779
BEGIN DESCRIPTION:
Mapping XS da05a281
END DESCRIPTION:
XS GIS Cut Line= 3
      1667713.38      7008410.27      1668720.32      7010076.92
      1669384.37      7010979.68
#Sta/Elev= 30
  3055.7 1605.67  3134.8 1593.21  3265.5 1590.28  3296.6 1580.93  3354.8 1579.16
  3477.0 1566.24  3556.6 1570.84  3826.3 1573.07  3958.3 1568.40  4032.0 1561.18
  4147.8 1554.77  4746.1 1546.75  4869.6 1542.08  4957.4 1536.95  4997.1 1526.13
  4997.9 1525.63  5032.6 1526.13  5056.6 1533.80  5106.7 1538.26  5200.8 1538.56
  5264.9 1562.77  5307.3 1572.03  5321.9 1571.30  5328.1 1574.83  5336.6 1573.93
  5357.4 1578.76  5524.7 1591.66  5828.2 1602.70  6009.3 1608.48  6123.6 1615.87
#Mann=7,-1,0
  3055.7    0.07       0  4147.8   0.035       0  4869.6    0.07       0
  4997.1    0.07       0  5032.6    0.07       0  5524.7   0.035       0
  5828.2    0.07       0
Bank Sta=4997.1,5032.6
Exp/Cntr=0.3,0.1

Type RM Length L Ch R = 1,20605,742,742,742
BEGIN DESCRIPTION:
Mapping XS 2d77e53a
END DESCRIPTION:
XS GIS Cut Line= 3
      1667487.69      7008518.78      1668182.13      7010593.42
      1667978.14      7011813.00
#Sta/Elev= 30
  2817.7 1618.18  2892.0 1608.06  3049.8 1596.88  3334.0 1585.17  3432.5 1583.29
  3486.5 1580.94  3530.1 1575.50  3676.0 1570.12  3791.5 1551.31  4469.3 1542.77
  4609.9 1541.56  4681.4 1538.34  4799.4 1536.27  4933.5 1527.22  4970.3 1527.97
  4971.2 1525.07  4972.1 1524.57  5007.2 1525.07  5010.3 1532.95  5016.8 1537.01
  5060.8 1554.72  5077.5 1557.90  5253.5 1561.43  5320.4 1570.55  5566.6 1583.58
  5793.7 1592.17  5902.3 1593.12  5936.2 1595.60  6165.5 1601.22  6242.0 1605.48
#Mann=12,-1,0
  2817.7    0.07       0  3432.5   0.035       0  3530.1    0.07       0
  3791.5   0.035       0  4469.3    0.07       0  4609.9   0.035       0
  4681.4    0.07       0  4971.2    0.07       0  5007.2    0.07       0
  5566.6   0.035       0  5793.7    0.07       0  5936.2   0.035       0
Bank Sta=4971.2,5007.2
Exp/Cntr=0.3,0.1

Type RM Length L Ch R = 1,19863,1029,1029,1029
BEGIN DESCRIPTION:
Mapping XS b40c52b0
END DESCRIPTION:
XS GIS Cut Line= 3
      1667228.13      7008537.85      1667488.55      7010454.53
      1667493.76      7011980.53
#Sta/Elev= 30
  3082.2 1652.69  3102.5 1646.50  3241.7 1629.50  3294.3 1619.99  3486.0 1597.35
  3809.0 1577.75  3980.5 1540.94  4209.0 1539.71  4665.2 1538.87  4798.0 1535.14
  4808.8 1537.62  4838.3 1532.33  4919.1 1530.85  4948.6 1524.81  4997.7 1521.67
  4998.6 1521.17  5033.7 1521.67  5040.0 1528.26  5060.0 1537.52  5086.7 1545.99
  5120.0 1555.05  5216.1 1559.20  5270.0 1556.83  5320.2 1560.73  5416.2 1567.75
  6183.3 1596.76  6277.6 1602.18  6289.3 1602.88  6460.0 1615.18  6542.5 1626.48
#Mann=12,-1,0
  3082.2    0.07       0  4209.0   0.035       0  4665.2    0.07       0
  4997.7    0.07       0  5033.7    0.07       0  5086.7    0.07       0
  5216.1   0.035       0  5320.2    0.07       0  5416.2   0.035       0
  6183.3    0.07       0  6277.6   0.035       0  6289.3    0.07       0
Bank Sta=4997.7,5033.7
Exp/Cntr=0.3,0.1

Type RM Length L Ch R = 1,18834,909,909,909
BEGIN DESCRIPTION:
Mapping XS 7b1f86de
END DESCRIPTION:
XS GIS Cut Line= 3
      1666991.16      7008681.07      1666648.27      7009957.13
      1666205.58      7011597.72
#Sta/Elev= 30
  3699.5 1652.63  3768.8 1648.03  3817.5 1639.78  3897.4 1632.25  4100.2 1597.67
  4234.8 1587.25  4321.7 1576.13  4421.2 1543.79  4471.2 1533.70  4619.8 1531.27
  4785.9 1528.58  4820.7 1519.25  4833.5 1518.71  4896.5 1523.44  4970.0 1521.53
  5000.6 1517.85  5001.4 1517.35  5036.8 1517.85  5039.1 1519.21  5055.3 1524.17
  5090.0 1526.77  5104.6 1535.19  5129.9 1539.81  5319.1 1542.74  5513.5 1564.72
  5600.8 1567.36  6016.5 1573.47  6089.1 1574.97  6228.0 1578.70  6720.1 1597.37
#Mann=11,-1,0
  3699.5    0.07       0  4619.8   0.035       0  4833.5    0.07       0
  4896.5   0.035       0  5000.6   0.035       0  5036.8   0.035       0
  5039.1    0.07       0  5600.8   0.035       0  6016.5    0.07       0
  6089.1   0.035       0  6228.0    0.07       0
Bank Sta=5000.6,5036.8
Exp/Cntr=0.3,0.1

Type RM Length L Ch R = 1,17925,809,809,809
BEGIN DESCRIPTION:
Mapping XS e2433cb1
END DESCRIPTION:
XS GIS Cut Line= 3
      1666465.99      7008355.56      1666005.91      7009345.15
      1665138.43      7011184.21
#Sta/Elev= 30
  3919.8 1612.04  4028.1 1597.32  4176.4 1588.34  4308.2 1569.43  4405.3 1571.02
  4410.8 1568.87  4479.5 1574.68  4688.9 1577.83  4788.1 1573.14  4839.3 1556.60
  4870.9 1538.82  4919.4 1524.03  4953.8 1517.12  4964.0 1511.51  4964.8 1511.01
  5000.4 1511.51  5027.9 1512.67  5080.6 1522.65  5126.9 1526.18  5180.1 1526.57
  5261.2 1521.72  5511.7 1532.43  5676.7 1543.97  5925.0 1552.01  6020.4 1558.87
  6295.7 1570.14  6644.5 1582.13  6831.5 1594.39  7004.5 1621.73  7044.5 1632.04
#Mann=9,-1,0
  3919.8    0.07       0  4688.9    0.16       0  4919.4    0.07       0
  4964.0    0.07       0  5000.4    0.07       0  5126.9   0.035       0
  5925.0    0.07       0  6295.7   0.035       0  6644.5    0.07       0
Bank Sta=4964,5000.4
Exp/Cntr=0.3,0.1

Type RM Length L Ch R = 1,17116,657,657,657
BEGIN DESCRIPTION:
Mapping XS a52679a9
END DESCRIPTION:
XS GIS Cut Line= 3
      1666140.66      7008241.44      1665250.05      7009152.88
      1663969.81      7010552.83
#Sta/Elev= 30
  3748.3 1619.44  3870.0 1608.00  3954.9 1596.40  4322.7 1573.04  4527.7 1550.51
  4534.8 1547.01  4612.5 1549.15  4754.0 1541.05  4888.5 1525.44  4930.9 1515.46
  4997.4 1511.18  4998.3 1510.68  5034.1 1511.18  5051.1 1516.55  5107.9 1519.21
  5242.3 1517.27  5284.8 1523.81  5379.3 1530.43  5476.0 1532.28  5503.9 1526.77
  5546.3 1532.07  5646.9 1535.04  5705.7 1538.50  5871.5 1545.07  5978.1 1548.86
  6134.0 1562.46  6601.5 1581.52  6735.9 1597.35  6870.3 1620.32  6919.7 1633.97
#Mann=7,-1,0
  3748.3    0.07       0  4997.4    0.07       0  5034.1    0.07       0
  5379.3   0.035       0  5646.9    0.07       0  5705.7   0.035       0
  5871.5    0.07       0
Bank Sta=4997.4,5034.1
Exp/Cntr=0.3,0.1

Type RM Length L Ch R = 1,16459,580,580,580
BEGIN DESCRIPTION:
Mapping XS c02a8749
END DESCRIPTION:
XS GIS Cut Line= 3
      1665942.78      7008194.54      1664692.76      7008934.13
      1663558.66      7009891.36
#Sta/Elev= 30
  3551.9 1599.57  3983.0 1576.57  4061.5 1570.34  4152.6 1564.06  4327.8 1551.50
  4525.2 1543.40  4589.5 1530.83  4676.4 1521.81  4940.5 1515.96  4999.0 1506.15
  5001.2 1503.05  5002.1 1502.55  5038.0 1503.05  5040.7 1507.84  5062.4 1516.17
  5076.7 1521.46  5091.0 1523.37  5140.5 1520.88  5197.6 1525.19  5306.1 1527.12
  5482.9 1535.38  5629.5 1542.27  5715.2 1552.04  5778.9 1554.45  6119.5 1581.12
  6247.0 1600.73  6304.2 1612.06  6353.6 1617.89  6425.1 1636.30  6488.4 1647.49
#Mann=7,-1,0
  3551.9    0.07       0  4061.5    0.16       0  4152.6    0.07       0
  5001.2    0.07       0  5038.0    0.07       0  5306.1   0.035       0
  5482.9    0.07       0
Bank Sta=5001.2,5038
Exp/Cntr=0.3,0.1

Type RM Length L Ch R = 1,15879,616,616,616
BEGIN DESCRIPTION:
Mapping XS ad848e4a
END DESCRIPTION:
XS GIS Cut Line= 3
      1665752.63      7007811.75      1664351.62      7008483.61
      1663456.04      7009103.22
#Sta/Elev= 30
  3452.5 1581.15  3575.7 1580.82  3761.8 1579.11  3831.0 1577.90  3942.4 1573.66
  4146.1 1555.15  4287.6 1545.89  4429.0 1541.54  4525.6 1524.59  4565.0 1520.09
  4799.6 1515.86  4813.0 1515.34  4893.2 1514.33  4947.1 1504.14  4982.5 1502.86
  4983.4 1502.36  5019.4 1502.86  5021.6 1515.05  5027.7 1518.45  5183.6 1524.69
  5215.9 1525.60  5302.3 1528.54  5430.4 1535.42  5540.6 1553.57  5582.5 1561.19
  5639.3 1565.58  5669.0 1570.86  5761.6 1576.09  5919.7 1590.53  6095.3 1619.76
#Mann=13,-1,0
  3452.5    0.07       0  3575.7   0.035       0  3761.8    0.07       0
  3831.0    0.16       0  3942.4    0.07       0  4799.6    0.16       0
  4813.0    0.07       0  4982.5    0.07       0  5019.4    0.07       0
  5183.6   0.035       0  5215.9    0.07       0  5302.3   0.035       0
  5540.6    0.07       0
Bank Sta=4982.5,5019.4
Exp/Cntr=0.3,0.1

Type RM Length L Ch R = 1,15263,646,646,646
BEGIN DESCRIPTION:
Mapping XS cf86985e
END DESCRIPTION:
XS GIS Cut Line= 3
      1665185.66      7006989.84      1664109.26      7007944.72
      1663425.21      7008722.51
#Sta/Elev= 30
  3565.1 1573.49  3584.0 1571.94  3685.0 1565.55  3989.4 1531.07  4260.3 1519.95
  4329.0 1514.60  4366.9 1516.83  4747.1 1514.01  4804.0 1510.00  4896.0 1512.39
  4916.9 1509.81  4931.1 1504.18  4959.6 1502.66  4967.1 1504.49  4969.5 1502.03
  4970.4 1501.53  5006.5 1502.03  5009.5 1504.27  5030.8 1505.78  5065.9 1525.95
  5154.2 1527.57  5190.5 1527.88  5378.0 1532.98  5441.6 1539.06  5533.6 1554.78
  5576.3 1557.62  5611.4 1563.68  5845.8 1577.87  5958.7 1587.76  6039.8 1597.42
#Mann=8,-1,0
  3565.1    0.16       0  3584.0    0.07       0  4260.3   0.035       0
  4366.9    0.07       0  4969.5    0.07       0  5006.5    0.07       0
  5154.2   0.035       0  5190.5    0.07       0
Bank Sta=4969.5,5006.5
Exp/Cntr=0.3,0.1

Type RM Length L Ch R = 1,14617,486,486,486
BEGIN DESCRIPTION:
Mapping XS 481e7592
END DESCRIPTION:
XS GIS Cut Line= 3
      1664923.47      7006819.73      1664046.76      7007349.23
      1663230.79      7008078.39
#Sta/Elev= 30
  3983.2 1571.72  4068.0 1564.46  4242.6 1532.75  4414.3 1525.02  4422.4 1524.62
  4542.4 1520.80  4767.3 1515.13  4978.1 1510.41  4986.1 1506.01  4986.7 1498.18
  4987.7 1497.68  5024.3 1498.18  5036.5 1502.47  5057.4 1505.20  5142.7 1504.55
  5277.2 1507.54  5291.4 1508.83  5298.2 1511.78  5304.9 1510.82  5312.4 1513.94
  5319.1 1512.64  5326.6 1516.00  5333.3 1514.41  5355.0 1519.35  5418.5 1525.54
  5432.7 1529.83  5475.4 1534.24  5659.3 1543.39  5942.7 1567.42  6101.7 1575.28
#Mann=7,-1,0
  3983.2    0.07       0  4414.3   0.035       0  4422.4    0.07       0
  4542.4   0.035       0  4767.3    0.07       0  4986.7    0.07       0
  5024.3    0.07       0
Bank Sta=4986.7,5024.3
Exp/Cntr=0.3,0.1

Type RM Length L Ch R = 1,14131,495,495,495
BEGIN DESCRIPTION:
Mapping XS a31fc025
END DESCRIPTION:
XS GIS Cut Line= 3
      1664489.45      7006403.07      1663734.26      7006988.99
      1662996.64      7008043.35
#Sta/Elev= 30
  4060.0 1544.82  4173.6 1542.56  4294.0 1529.62  4352.6 1526.66  4378.5 1525.93
  4522.1 1521.91  4686.0 1513.40  4893.3 1512.57  4922.2 1508.41  4928.6 1503.12
  4972.0 1502.93  4978.3 1499.75  5001.0 1497.14  5009.2 1493.07  5010.2 1492.57
  5046.9 1493.07  5051.2 1497.21  5063.8 1503.15  5078.7 1506.44  5158.5 1507.85
  5342.3 1512.03  5417.4 1515.46  5459.7 1520.90  5510.3 1531.12  5558.6 1534.87
  5594.3 1536.48  5703.9 1543.23  5826.0 1557.53  6022.3 1569.48  6302.6 1578.48
#Mann=10,-1,0
  4060.0    0.07       0  4352.6   0.035       0  4378.5    0.07       0
  5009.2    0.07       0  5046.9    0.07       0  5158.5   0.035       0
  5342.3    0.07       0  5558.6   0.035       0  5594.3    0.07       0
  6022.3   0.035       0
Bank Sta=5009.2,5046.9
Exp/Cntr=0.3,0.1

Type RM Length L Ch R = 1,13636,281,281,281
BEGIN DESCRIPTION:
Mapping XS d15ac262
END DESCRIPTION:
XS GIS Cut Line= 3
      1663834.07      7006550.63      1663321.93      7006763.30
      1662727.32      7008039.32
#Sta/Elev= 30
  4451.9 1521.57  4538.0 1520.68  4644.8 1519.93  4850.9 1518.13  4900.8 1516.05
  4916.5 1512.97  4930.1 1507.25  4966.6 1497.58  4977.8 1496.69  4983.2 1493.51
  4995.2 1490.88  4996.2 1490.38  5032.9 1490.88  5054.3 1497.34  5088.9 1502.30
  5159.3 1506.18  5170.3 1506.62  5232.3 1508.58  5265.4 1507.19  5294.0 1509.61
  5413.9 1512.64  5465.2 1519.41  5505.4 1527.05  5533.8 1535.09  5596.3 1541.92
  5676.5 1555.82  5806.0 1566.22  5912.5 1568.40  6361.8 1575.44  6414.2 1574.64
#Mann=10,-1,0
  4451.9    0.07       0  4538.0   0.035       0  4644.8    0.07       0
  4850.9    0.16       0  4966.6    0.07       0  4995.2    0.07       0
  5032.9    0.07       0  5159.3   0.035       0  5170.3    0.07       0
  5912.5   0.035       0
Bank Sta=4995.2,5032.9
Exp/Cntr=0.3,0.1

Type RM Length L Ch R = 1,13355,266,266,266
BEGIN DESCRIPTION:
Mapping XS 0f837413
END DESCRIPTION:
XS GIS Cut Line= 3
      1663453.74      7006384.09      1663068.28      7006668.84
      1662659.39      7007361.88
#Sta/Elev= 30
  4533.4 1518.43  4744.5 1516.58  4864.7 1514.14  4900.2 1511.63  4906.4 1508.86
  4914.8 1507.79  4921.1 1503.34  4935.7 1500.27  4964.9 1498.98  4971.2 1496.70
  4985.8 1495.29  4987.8 1492.27  4988.7 1491.77  5025.5 1492.27  5034.9 1494.80
  5058.1 1494.52  5087.5 1497.53  5116.1 1498.00  5146.1 1502.46  5306.1 1505.01
  5358.8 1507.48  5386.1 1510.47  5410.4 1515.60  5452.9 1524.84  5489.0 1536.76
  5518.8 1547.40  5569.0 1560.87  5604.6 1563.76  5673.0 1564.91  5817.3 1561.03
#Mann=6,-1,0
  4533.4   0.035       0  4744.5    0.07       0  4987.8    0.07       0
  5025.5    0.07       0  5410.4   0.035       0  5489.0    0.07       0
Bank Sta=4987.8,5025.5
Exp/Cntr=0.3,0.1

Type RM Length L Ch R = 1,13089,398,398,398
BEGIN DESCRIPTION:
Mapping XS ed915a54
END DESCRIPTION:
XS GIS Cut Line= 3
      1663166.17      7006480.04      1662811.99      7006641.50
      1662557.50      7007194.62
#Sta/Elev= 30
  4619.2 1514.36  4821.5 1513.39  4839.0 1511.82  4844.5 1508.86  4862.1 1509.10
  4867.6 1504.38  4890.6 1504.63  4896.1 1500.40  4913.7 1499.75  4919.2 1494.39
  4928.2 1494.93  4931.3 1490.39  4932.3 1489.89  4969.0 1490.39  4988.3 1492.40
  5040.1 1491.62  5103.5 1498.43  5147.7 1496.94  5169.7 1500.89  5246.8 1503.75
  5268.8 1505.89  5298.3 1511.35  5326.8 1518.75  5334.8 1522.53  5372.7 1533.63
  5378.9 1537.55  5401.2 1545.86  5424.2 1552.31  5441.6 1555.62  5617.3 1556.39
#Mann=3,-1,0
  4619.2    0.07       0  4931.3    0.07       0  4969.0    0.07       0
Bank Sta=4931.3,4969
Exp/Cntr=0.3,0.1

Type RM Length L Ch R = 1,12691,237,237,237
BEGIN DESCRIPTION:
Fish Creek 25.0
END DESCRIPTION:
XS GIS Cut Line= 3
      1663259.29      7006404.95      1662441.83      7006574.26
      1662148.13      7007227.91
#Sta/Elev= 30
  4165.2 1515.64  4323.5 1513.76  4363.6 1514.37  4450.9 1511.12  4551.3 1509.93
  4651.7 1506.45  4772.1 1500.15  4812.9 1501.62  4842.2 1499.79  4874.2 1495.76
  4892.4 1495.06  4897.5 1493.13  4956.3 1490.52  4967.7 1490.38  4968.7 1489.88
  5005.4 1490.38  5027.9 1490.91  5053.4 1492.59  5076.5 1496.67  5105.2 1498.47
  5122.8 1502.24  5151.5 1504.30  5174.6 1511.04  5190.5 1514.23  5234.3 1527.67
  5256.3 1532.65  5376.8 1538.76  5481.8 1540.31  5613.5 1541.37  5716.6 1540.60
#Mann=7,-1,0
  4165.2   0.035       0  4323.5    0.07       0  4956.3   0.035       0
  4967.7   0.035       0  5005.4   0.035       0  5027.9    0.07       0
  5481.8   0.035       0
Bank Sta=4967.7,5005.4
Exp/Cntr=0.3,0.1

Type RM Length L Ch R = 1,12454,319,319,319
BEGIN DESCRIPTION:
Mapping XS e6801966
END DESCRIPTION:
XS GIS Cut Line= 3
      1661922.99      7005752.03      1662253.73      7006442.14
      1662071.43      7007158.33
#Sta/Elev= 30
  4234.9 1561.78  4277.3 1557.93  4345.3 1544.16  4407.7 1525.94  4435.9 1519.69
  4481.2 1513.48  4594.5 1504.02  4607.5 1499.10  4696.2 1505.44  4758.7 1501.17
  4786.9 1502.12  4818.2 1496.38  4862.5 1496.09  4872.0 1493.64  4877.5 1494.98
  4884.7 1491.05  4894.6 1490.15  4954.5 1491.95  4995.9 1489.59  4998.7 1487.89
  4999.7 1487.39  5038.3 1487.89  5047.5 1493.08  5078.4 1497.42  5171.3 1499.61
  5198.6 1504.21  5315.8 1531.07  5417.2 1537.31  5523.2 1538.40  5739.2 1538.46
#Mann=6,-1,0
  4234.9    0.07       0  4954.5   0.035       0  4998.7   0.035       0
  5038.3   0.035       0  5198.6    0.07       0  5523.2   0.035       0
Bank Sta=4998.7,5038.3
Exp/Cntr=0.3,0.1

Type RM Length L Ch R = 1,12135,296,296,296
BEGIN DESCRIPTION:
Mapping XS b94b7e8a
END DESCRIPTION:
XS GIS Cut Line= 3
      1661795.38      7005858.78      1661967.27      7006340.58
      1661943.83      7007022.83
#Sta/Elev= 30
  4491.3 1545.70  4522.3 1539.26  4562.0 1526.51  4567.3 1526.36  4592.8 1519.22
  4623.6 1513.02  4654.4 1510.27  4692.2 1503.45  4724.1 1500.67  4883.3 1494.19
  4904.6 1489.99  4951.9 1487.09  4957.6 1488.79  4977.4 1487.56  4979.0 1485.37
  4980.0 1484.87  5018.7 1485.37  5020.3 1487.30  5030.3 1491.04  5050.3 1495.59
  5090.3 1494.22  5190.4 1497.27  5215.0 1501.83  5220.4 1504.43  5280.4 1517.91
  5330.5 1522.93  5390.5 1532.12  5427.7 1534.14  5570.6 1536.36  5685.5 1536.73
#Mann=5,-1,0
  4491.3    0.07       0  4979.0    0.07       0  5018.7    0.07       0
  5427.7   0.035       0  5570.6    0.07       0
Bank Sta=4979,5018.7
Exp/Cntr=0.3,0.1

Type RM Length L Ch R = 1,11839,375,375,375
BEGIN DESCRIPTION:
Mapping XS 38b847c0
END DESCRIPTION:
XS GIS Cut Line= 3
      1661574.05      7005806.76      1661688.62      7006296.31
      1661792.79      7007007.24
#Sta/Elev= 30
  4505.4 1561.88  4537.5 1559.93  4547.8 1557.78  4599.1 1543.63  4622.0 1539.21
  4707.0 1514.54  4754.6 1509.25  4792.0 1499.71  4814.8 1495.99  4876.4 1494.20
  4929.7 1489.14  4958.6 1484.88  4975.5 1485.29  4979.1 1485.69  4979.8 1484.52
  4980.8 1484.02  5019.5 1484.52  5030.1 1490.05  5040.2 1492.86  5191.8 1494.35
  5220.8 1500.14  5225.9 1499.58  5232.2 1502.17  5250.9 1504.08  5313.1 1505.48
  5365.6 1508.46  5424.3 1514.39  5454.6 1519.14  5626.4 1532.60  5726.7 1534.03
#Mann=5,-1,0
  4505.4    0.07       0  4975.5   0.035       0  4979.8   0.035       0
  5019.5   0.035       0  5250.9    0.07       0
Bank Sta=4979.8,5019.5
Exp/Cntr=0.3,0.1

Type RM Length L Ch R = 1,11464,348,348,348
BEGIN DESCRIPTION:
Mapping XS 8cc81690
END DESCRIPTION:
XS GIS Cut Line= 3
      1661276.88      7005861.39      1661344.15      7006191.24
      1661690.68      7006966.59
#Sta/Elev= 30
  4666.8 1550.49  4704.2 1553.03  4724.6 1552.33  4731.1 1549.55  4736.2 1549.93
  4781.6 1534.00  4786.7 1534.17  4796.0 1528.85  4816.4 1521.56  4882.7 1507.32
  4908.3 1498.31  4978.6 1487.54  4979.4 1480.29  4980.4 1479.79  5019.1 1480.29
  5022.5 1482.80  5032.7 1484.07  5115.4 1491.60  5175.1 1490.14  5229.9 1491.25
  5242.3 1492.95  5255.6 1497.92  5273.7 1502.68  5420.8 1503.14  5504.3 1503.81
  5598.0 1506.68  5689.9 1518.04  5744.7 1521.78  5810.4 1529.36  5852.7 1531.10
#Mann=7,-1,0
  4666.8    0.07       0  4979.4    0.07       0  5019.1    0.07       0
  5255.6   0.035       0  5420.8    0.07       0  5504.3   0.035       0
  5598.0    0.07       0
Bank Sta=4979.4,5019.1
Exp/Cntr=0.3,0.1

Type RM Length L Ch R = 1,11116,355,355,355
BEGIN DESCRIPTION:
Mapping XS fb61af78
END DESCRIPTION:
XS GIS Cut Line= 3
      1660753.89      7005902.63      1661012.12      7006241.15
      1661569.08      7007004.00
#Sta/Elev= 30
  4575.7 1548.45  4630.9 1543.96  4751.5 1525.44  4766.0 1525.11  4786.8 1518.46
  4830.4 1510.48  4851.2 1502.75  4865.8 1502.00  4872.0 1498.61  4909.4 1489.05
  4965.5 1488.24  5009.3 1483.55  5095.0 1486.29  5095.9 1483.54  5096.9 1483.04
  5135.8 1483.54  5136.8 1485.15  5172.3 1488.08  5222.5 1489.16  5266.5 1498.39
  5309.5 1499.34  5384.6 1499.46  5482.4 1500.07  5632.4 1500.05  5643.2 1500.19
  5716.0 1501.65  5789.4 1510.33  5831.1 1517.70  5911.9 1524.64  5946.0 1527.23
#Mann=9,-1,0
  4575.7    0.07       0  5095.9    0.07       0  5135.8    0.07       0
  5309.5   0.035       0  5384.6    0.07       0  5482.4   0.035       0
  5632.4    0.07       0  5643.2   0.035       0  5911.9    0.07       0
Bank Sta=5095.9,5135.8
Exp/Cntr=0.3,0.1

Type RM Length L Ch R = 1,10761,237,237,237
BEGIN DESCRIPTION:
Mapping XS b341b6e1
END DESCRIPTION:
XS GIS Cut Line= 3
      1660560.30      7006064.08      1660771.23      7006472.92
      1661460.71      7006917.83
#Sta/Elev= 30
  4540.6 1547.52  4556.2 1546.22  4561.8 1548.87  4578.3 1545.87  4584.0 1547.58
  4590.0 1545.68  4657.5 1545.30  4694.8 1542.31  4761.2 1531.82  4849.9 1501.51
  4894.2 1489.84  4955.0 1480.05  4977.2 1483.07  4993.7 1481.91  5028.9 1486.74
  5051.4 1486.01  5057.4 1484.87  5058.6 1475.86  5059.6 1475.36  5098.5 1475.86
  5100.3 1480.05  5114.8 1486.58  5130.0 1491.45  5151.1 1493.57  5290.3 1497.88
  5456.3 1498.23  5604.6 1498.56  5706.1 1499.65  5758.9 1502.84  5821.2 1512.63
#Mann=6,-1,0
  4540.6    0.07       0  5058.6    0.07       0  5098.5    0.07       0
  5456.3   0.035       0  5604.6    0.07       0  5706.1   0.035       0
Bank Sta=5058.6,5098.5
Exp/Cntr=0.3,0.1

Type RM Length L Ch R = 1,10524,263,263,263
BEGIN DESCRIPTION:
Mapping XS 68e95a91
END DESCRIPTION:
XS GIS Cut Line= 3
      1660226.95      7006717.72      1660755.61      7006704.70
      1661487.37      7006988.55
#Sta/Elev= 30
  4471.8 1589.86  4489.9 1585.22  4539.9 1578.25  4601.2 1566.75  4606.8 1565.82
  4649.9 1560.26  4679.9 1551.95  4759.9 1515.74  4809.9 1496.77  4830.0 1491.56
  4850.0 1481.89  4860.0 1480.27  4930.0 1482.37  4940.0 1481.53  4949.7 1476.87
  4950.7 1476.37  4990.3 1476.87  5010.7 1480.18  5032.1 1487.95  5074.3 1492.68
  5109.6 1491.67  5169.1 1494.27  5231.0 1496.24  5361.2 1496.78  5545.3 1497.96
  5592.6 1496.37  5635.6 1498.01  5689.5 1502.90  5768.5 1517.97  5785.5 1519.51
#Mann=10,-1,0
  4471.8    0.07       0  4601.2   0.035       0  4606.8    0.07       0
  4949.7    0.07       0  4990.3    0.07       0  5169.1   0.035       0
  5231.0    0.07       0  5361.2   0.035       0  5592.6    0.07       0
  5635.6   0.035       0
Bank Sta=4949.7,4990.3
Exp/Cntr=0.3,0.1

Type RM Length L Ch R = 1,10261,209,209,209
BEGIN DESCRIPTION:
Mapping XS a1c29fe4
END DESCRIPTION:
XS GIS Cut Line= 3
      1660315.49      7006954.69      1660753.01      7006967.72
      1661510.39      7007040.59
#Sta/Elev= 30
  4560.3 1595.49  4589.8 1586.83  4639.8 1576.79  4679.9 1564.36  4697.6 1561.77
  4711.6 1559.51  4749.9 1546.96  4769.9 1536.28  4829.9 1511.27  4837.2 1508.64
  4842.2 1509.98  4859.9 1500.13  4900.0 1483.18  4939.7 1474.52  4940.7 1474.02
  4980.3 1474.52  4990.0 1478.13  5001.5 1474.56  5054.2 1480.23  5070.3 1484.06
  5110.4 1487.12  5214.6 1489.61  5311.4 1494.34  5442.7 1494.74  5512.4 1494.22
  5592.7 1497.71  5663.1 1506.65  5703.2 1516.13  5734.8 1520.50  5758.9 1523.92
#Mann=9,-1,0
  4560.3    0.07       0  4697.6   0.035       0  4711.6    0.07       0
  4939.7    0.07       0  4980.3    0.07       0  5110.4   0.035       0
  5214.6    0.07       0  5442.7   0.035       0  5734.8    0.07       0
Bank Sta=4939.7,4980.3
Exp/Cntr=0.3,0.1

Type RM Length L Ch R = 1,10052,503,503,503
BEGIN DESCRIPTION:
Mapping XS c6ddb96f
END DESCRIPTION:
XS GIS Cut Line= 3
      1660336.34      7007220.32      1660758.21      7007176.05
      1661638.38      7007071.89
#Sta/Elev= 30
  4578.0 1565.11  4627.8 1561.21  4677.2 1558.93  4777.7 1548.20  4836.4 1533.14
  4841.4 1533.77  4873.7 1522.29  4918.5 1504.41  4958.7 1483.20  4978.8 1477.65
  5002.2 1475.15  5010.9 1472.20  5011.9 1471.70  5051.5 1472.20  5059.4 1475.84
  5089.6 1479.98  5139.9 1484.18  5321.2 1488.82  5372.5 1493.76  5405.1 1493.14
  5442.0 1492.15  5533.6 1494.65  5583.0 1496.75  5626.6 1501.70  5673.6 1509.36
  5696.6 1515.41  5791.7 1526.80  5855.7 1528.45  5862.6 1528.52  5888.5 1529.20
#Mann=11,-1,0
  4578.0    0.07       0  4627.8   0.035       0  4873.7    0.07       0
  5010.9    0.07       0  5051.5    0.07       0  5405.1   0.035       0
  5533.6    0.07       0  5626.6   0.035       0  5696.6    0.07       0
  5855.7   0.035       0  5862.6    0.07       0
Bank Sta=5010.9,5051.5
Exp/Cntr=0.3,0.1

Type RM Length L Ch R = 1,9549,580,580,580
BEGIN DESCRIPTION:
Mapping XS 6c09707a
END DESCRIPTION:
XS GIS Cut Line= 3
      1659939.47      7007444.89      1660907.35      7007631.52
      1662018.44      7007848.53
#Sta/Elev= 30
  4014.4 1567.24  4056.5 1567.92  4061.6 1565.91  4305.2 1560.14  4417.2 1550.83
  4458.0 1545.19  4533.5 1530.81  4590.4 1516.04  4682.0 1503.47  4702.4 1499.01
  4863.4 1489.75  4906.7 1486.14  4936.6 1476.15  4955.5 1474.03  4967.2 1470.87
  4968.2 1470.37  5007.8 1470.87  5038.5 1475.51  5120.0 1476.76  5150.6 1480.38
  5219.3 1481.77  5342.9 1484.76  5497.0 1489.64  5517.4 1487.10  5582.6 1503.66
  5609.1 1512.90  5660.0 1524.48  5731.3 1525.42  5845.5 1532.82  6132.2 1539.44
#Mann=7,-1,0
  4014.4    0.07       0  4863.4   0.035       0  4955.5    0.07       0
  4967.2    0.07       0  5007.8    0.07       0  5219.3   0.035       0
  5342.9    0.07       0
Bank Sta=4967.2,5007.8
Exp/Cntr=0.3,0.1

Type RM Length L Ch R = 1,8969,331,331,331
BEGIN DESCRIPTION:
Mapping XS ee8815a9
END DESCRIPTION:
XS GIS Cut Line= 3
      1659926.47      7007687.95      1661011.51      7008182.73
      1662111.93      7008148.07
#Sta/Elev= 30
  3814.5 1550.98  3841.8 1551.32  4087.0 1548.78  4184.6 1528.45  4241.7 1513.20
  4333.9 1497.50  4380.0 1492.75  4541.0 1484.53  4757.8 1481.33  4937.4 1478.63
  4960.4 1475.25  4966.9 1472.28  4968.6 1468.73  4969.6 1468.23  5009.3 1468.73
  5011.3 1470.93  5020.5 1469.23  5040.5 1474.15  5110.6 1469.00  5130.6 1469.82
  5190.6 1478.02  5230.6 1485.78  5316.0 1517.90  5321.0 1516.88  5340.7 1523.49
  5380.7 1530.86  5460.7 1532.98  5740.9 1528.61  5981.0 1541.10  6108.0 1552.43
#Mann=6,-1,0
  3814.5   0.035       0  3841.8    0.07       0  4541.0   0.035       0
  4757.8    0.07       0  4968.6    0.07       0  5009.3    0.07       0
Bank Sta=4968.6,5009.3
Exp/Cntr=0.3,0.1

Type RM Length L Ch R = 1,8638,362,362,362
BEGIN DESCRIPTION:
Mapping XS 21086214
END DESCRIPTION:
XS GIS Cut Line= 3
      1659323.16      7007813.82      1660950.75      7008495.23
      1662170.20      7008768.63
#Sta/Elev= 30
  3239.5 1574.55  3269.2 1569.72  3337.3 1557.86  3549.3 1543.65  3688.0 1525.82
  3732.1 1516.79  3771.6 1503.61  3808.9 1499.05  3832.6 1506.49  3885.6 1507.09
  3909.4 1511.07  4039.2 1509.42  4228.0 1487.06  4386.0 1481.19  4841.7 1477.74
  4937.1 1473.06  4998.2 1466.23  4999.2 1465.73  5038.9 1466.23  5110.8 1475.11
  5182.6 1506.22  5225.5 1511.58  5317.3 1515.36  5377.3 1509.11  5490.0 1527.82
  5520.7 1525.60  5561.7 1532.12  5623.2 1531.01  5819.8 1548.72  6253.7 1565.40
#Mann=8,-1,0
  3239.5   0.035       0  3269.2    0.07       0  3688.0   0.035       0
  3771.6    0.07       0  4386.0   0.035       0  4937.1    0.07       0
  4998.2    0.07       0  5038.9    0.07       0
Bank Sta=4998.2,5038.9
Exp/Cntr=0.3,0.1
