--- Post Oak Creek.prj (project) ---

Proj Title=Post Oak Creek Base Level Engineering
Current Plan=p01
Default Exp/Contr=0.3,0.1
English Units
Geom File=g01
Flow File=f01
Plan File=p01
Y Axis Title=Elevation
X Axis Title(PF)=Main Channel Distance
X Axis Title(XS)=Station
BEGIN DESCRIPTION:
Post Oak Creek
END DESCRIPTION:
DSS Export Rating Curves= 0
DSS Export Rating Curve Sorted= 0
DSS Export Volume Flow Curves= 0
DXF OffsetX= 0
DXF OffsetY= 0
DXF ScaleX= 1
DXF ScaleY= 10

--- Post Oak Creek.p01 (plan) ---

Plan Title=Multiple Run
Short Identifier=Multiple
Geom File=g01
Flow File=f01
Subcritical Flow
K Sum by GR= 0
Std Step Tol= 0.01
Critical Tol= 0.01
Num of Std Step Trials= 20
Max Error Tol= 0.3
Flow Tol Ratio= 0.001
Split Flow NTrial= 30
Split Flow Tol= 0.02
Split Flow Ratio= 0.02
Log Output Level= 0
Friction Slope Method= 1
Unsteady Friction Slope Method= 2
Unsteady Bridges Friction Slope Method= 1
Parabolic Critical Depth
Global Vel Dist=  1 , 1 , 1
Global Log Level= 0
CheckData=True
Encroach Param= -1, 0, 0, 0
BEGIN DESCRIPTION:
Multiple Run
END DESCRIPTION:

--- Post Oak Creek.f01 (steady flow) ---

Flow Title=Multiple
Number of Profiles=7
Profile Names=10-year,25-year,50-year,1pct_min,100-year,1pct_plu,500-year
River Rch & RM= Post Oak Creek,Reach-1,27095
     176     236     283     169     337     673     485
River Rch & RM= Post Oak Creek,Reach-1,25833
     232     314     380     229     457     913     670
River Rch & RM= Post Oak Creek,Reach-1,22912
     419     589     731     451     899    1794    1378
River Rch & RM= Post Oak Creek,Reach-1,18358
     651     931    1170     729    1454    2901    2278
River Rch & RM= Post Oak Creek,Reach-1,14561
     643     915    1145     710    1416    2826    2199
River Rch & RM= Post Oak Creek,Reach-1,10002
     675     961    1203     746    1489    2971    2313
River Rch & RM= Post Oak Creek,Reach-1,6963
     819    1172    1471     915    1826    3643    2850
Boundary for River Rch & Prof#=Post Oak Creek,Reach-1,1
Up Type=0
Dn Type=3
Dn Slope=0.005
Boundary for River Rch & Prof#=Post Oak Creek,Reach-1,2
Up Type=0
Dn Type=3
Dn Slope=0.005
Boundary for River Rch & Prof#=Post Oak Creek,Reach-1,3
Up Type=0
Dn Type=3
Dn Slope=0.005
Boundary for River Rch & Prof#=Post Oak Creek,Reach-1,4
Up Type=0
Dn Type=3
Dn Slope=0.005
Boundary for River Rch & Prof#=Post Oak Creek,Reach-1,5
Up Type=0
Dn Type=3
Dn Slope=0.005
Boundary for River Rch & Prof#=Post Oak Creek,Reach-1,6
Up Type=0
Dn Type=3
Dn Slope=0.005
Boundary for River Rch & Prof#=Post Oak Creek,Reach-1,7
Up Type=0
Dn Type=3
Dn Slope=0.005

--- Post Oak Creek.g01 (geometry) ---

Geom Title=Existing Conditions

River Reach=Post Oak Creek,Reach-1
Reach XY= 30
      1613505.00      6986888.00      1613897.50      6986291.13
      1613554.95      6986003.34      1614153.03      6984932.35
      1613961.88      6983938.03      1614237.86      6983404.28
      1614725.04      6983137.39      1615157.28      6983432.95
      1616071.67      6982871.35      1616715.34      6982038.81
      1617502.55      6982682.55      1617807.43      6982632.48
      1619145.20      6981048.48      1620132.01      6980911.52
      1620410.18      6979943.44      1621138.98      6979638.24
      1621289.70      6980088.17      1621700.24      6979782.42
      1621748.33      6979246.95      1622397.54      6979581.95
      1622307.06      6979982.15      1622581.59      6980365.57
      1623434.79      6980838.52      1625106.64      6979691.14
      1625724.88      6979988.09      1626507.43      6979782.48
      1626760.24      6978990.09      1627599.12      6979039.96
      1628715.55      6979586.92      1629055.00      6979438.00

Type RM Length L Ch R = 1,27095,483,483,483
BEGIN DESCRIPTION:
Post Oak Creek 44.0
END DESCRIPTION:
XS GIS Cut Line= 3
      1614167.03      6987143.04      1613542.01      6986851.44
      1612726.07      6986601.38
#Sta/Elev= 30
  4310.3 1579.20  4354.4 1577.53  4422.9 1577.24  4594.1 1570.20  4707.8 1567.32
  4766.8 1566.02  4828.2 1565.45  4862.3 1563.73  4862.5 1563.23  4866.3 1563.73
  4930.7 1564.92  4976.4 1564.97  4998.2 1563.91  5031.1 1565.03  5100.4 1565.05
  5206.1 1565.26  5238.1 1566.41  5265.6 1565.56  5362.9 1566.82  5394.3 1568.38
  5434.6 1568.03  5488.4 1570.73  5510.6 1570.21  5570.9 1571.34  5603.5 1573.55
  5655.8 1573.69  5687.2 1576.23  5729.0 1576.23  5777.8 1578.84  5853.4 1580.13
#Mann=6,-1,0
  4310.3    0.07       0  4707.8   0.035       0  4766.8    0.07       0
  4862.3    0.07       0  4866.3    0.07       0  5100.4   0.045       0
Bank Sta=4862.3,4866.3
Exp/Cntr=0.3,0.1

Type RM Length L Ch R = 1,26612,619,619,619
BEGIN DESCRIPTION:
Mapping XS a5cedaad
END DESCRIPTION:
XS GIS Cut Line= 3
      1614221.75      6986814.71      1613669.68      6986470.96
      1612919.84      6986335.58
#Sta/Elev= 30
  4350.7 1573.02  4405.3 1571.81  4426.5 1570.33  4771.7 1564.68  4812.1 1564.25
  4925.7 1563.48  4947.7 1564.31  4999.0 1561.53  4999.3 1561.03  5003.0 1561.53
  5026.1 1563.60  5048.7 1563.51  5058.3 1564.43  5066.8 1566.28  5076.9 1566.80
  5097.2 1566.14  5117.6 1566.94  5137.9 1563.72  5158.5 1563.23  5310.6 1564.31
  5351.3 1566.24  5412.3 1566.37  5438.7 1568.20  5473.2 1567.93  5513.9 1570.11
  5564.7 1570.54  5604.5 1573.10  5656.1 1573.59  5696.8 1576.05  5763.0 1576.87
#Mann=7,-1,0
  4350.7    0.07       0  4771.7   0.035       0  4812.1    0.07       0
  4999.0    0.07       0  5003.0    0.07       0  5058.3   0.035       0
  5158.5   0.045       0
Bank Sta=4999,5003
Exp/Cntr=0.3,0.1

Type RM Length L Ch R = 1,25993,160,160,160
BEGIN DESCRIPTION:
Mapping XS b6853bab
END DESCRIPTION:
XS GIS Cut Line= 3
      1614497.79      6986171.49      1613638.43      6986179.30
      1612868.83      6986192.30
#Sta/Elev= 30
  4146.3 1573.11  4349.1 1569.37  4379.1 1569.65  4459.1 1566.67  4509.1 1562.02
  4599.1 1565.57  4839.1 1562.64  4859.1 1562.76  4869.1 1564.72  4879.1 1564.87
  4919.1 1559.47  4937.1 1558.20  4937.4 1557.70  4941.1 1558.20  4979.1 1560.56
  5059.1 1571.22  5069.1 1571.39  5099.1 1563.98  5109.1 1563.08  5169.1 1562.76
  5289.2 1564.52  5319.2 1566.33  5349.2 1566.30  5379.2 1567.92  5519.2 1571.11
  5549.2 1573.18  5599.2 1573.60  5639.2 1575.93  5689.2 1576.15  5775.4 1578.44
#Mann=3,-1,0
  4146.3   0.035       0  4937.1   0.035       0  4941.1   0.035       0
Bank Sta=4937.1,4941.1
Exp/Cntr=0.3,0.1

Type RM Length L Ch R = 1,25833,404,404,404
BEGIN DESCRIPTION:
Mapping XS c672449b
END DESCRIPTION:
XS GIS Cut Line= 3
      1614492.60      6986002.21      1613557.70      6986046.49
      1612885.80      6986054.30
#Sta/Elev= 30
  4070.8 1571.91  4145.1 1570.22  4238.6 1569.01  4278.6 1567.93  4301.2 1568.00
  4367.5 1565.98  4418.8 1564.94  4428.8 1563.73  4448.8 1562.62  4498.9 1561.80
  4538.9 1562.96  4579.0 1563.09  4724.1 1561.93  4919.4 1561.92  4933.7 1561.60
  4939.4 1560.76  4987.4 1560.31  4987.7 1559.81  4991.2 1559.81  4991.4 1560.31
  5019.5 1561.33  5059.5 1560.52  5089.5 1561.26  5159.5 1561.40  5209.5 1564.68
  5429.5 1572.28  5449.5 1573.50  5570.8 1575.57  5619.5 1577.31  5678.7 1578.18
#Mann=6,-1,0
  4070.8   0.035       0  4145.1    0.07       0  4367.5   0.035       0
  4724.1    0.07       0  4987.4    0.07       0  4991.4    0.07       0
Bank Sta=4987.4,4991.4
Exp/Cntr=0.3,0.1

Type RM Length L Ch R = 1,25429,524,524,524
BEGIN DESCRIPTION:
Mapping XS acf539b9
END DESCRIPTION:
XS GIS Cut Line= 3
      1614449.01      6985716.19      1613706.83      6985697.96
      1612941.19      6985752.65
#Sta/Elev= 30
  4257.2 1568.12  4279.7 1567.76  4341.2 1567.62  4401.3 1566.46  4541.3 1565.33
  4581.3 1564.01  4623.1 1564.19  4821.4 1559.49  4859.4 1557.92  4859.6 1557.42
  4863.1 1557.42  4863.4 1557.92  4920.3 1560.03  4961.4 1560.14  4991.4 1558.10
  4998.0 1559.16  5011.5 1559.81  5031.5 1563.16  5051.6 1559.71  5068.5 1558.26
  5111.7 1560.16  5161.8 1560.21  5332.3 1562.92  5494.6 1567.82  5592.9 1572.69
  5623.0 1573.08  5629.9 1573.73  5634.9 1573.40  5663.1 1574.73  5767.2 1575.93
#Mann=6,-1,0
  4257.2   0.035       0  4279.7    0.07       0  4623.1   0.035       0
  4859.4    0.07       0  4863.4   0.035       0  4920.3    0.07       0
Bank Sta=4859.4,4863.4
Exp/Cntr=0.3,0.1

Type RM Length L Ch R = 1,24905,575,575,575
BEGIN DESCRIPTION:
Mapping XS 368c1f5a
END DESCRIPTION:
XS GIS Cut Line= 3
      1614435.97      6985424.52      1613912.56      6985281.29
      1612790.11      6985487.03
#Sta/Elev= 30
  4456.9 1565.67  4458.3 1565.67  4497.4 1565.61  4520.1 1564.61  4582.3 1563.81
  4675.6 1563.81  4758.6 1563.18  4810.4 1561.73  4838.9 1562.13  4924.4 1559.74
  4955.7 1555.61  4956.0 1555.11  4960.0 1555.11  4960.3 1555.61  4986.7 1557.25
  5010.7 1557.41  5058.1 1559.34  5139.4 1559.65  5175.2 1558.37  5281.5 1558.16
  5312.2 1557.35  5352.9 1558.35  5495.2 1559.57  5668.1 1563.34  5688.4 1564.49
  5759.6 1565.96  5785.3 1567.45  5954.9 1572.40  5991.7 1572.18  6140.7 1572.92
#Mann=5,-1,0
  4456.9   0.035       0  4458.3    0.07       0  4955.7    0.07       0
  4960.3    0.07       0  5991.7   0.035       0
Bank Sta=4955.7,4960.3
Exp/Cntr=0.3,0.1

Type RM Length L Ch R = 1,24330,297,297,297
BEGIN DESCRIPTION:
Mapping XS 6cd703d5
END DESCRIPTION:
XS GIS Cut Line= 3
      1614643.74      6984959.34      1614151.16      6984844.34
      1612908.87      6985225.91
#Sta/Elev= 30
  4498.2 1565.78  4599.6 1563.93  4650.9 1563.87  4699.6 1561.35  4733.1 1561.27
  4765.7 1559.57  4948.7 1556.60  4997.1 1554.20  4997.5 1553.70  5001.8 1554.20
  5035.1 1555.52  5100.5 1556.26  5115.1 1554.94  5124.0 1555.05  5138.5 1556.13
  5177.9 1556.29  5198.7 1554.37  5219.7 1556.36  5307.3 1558.27  5340.0 1557.23
  5622.9 1556.95  5878.7 1559.41  6058.5 1563.25  6077.5 1564.05  6086.0 1565.24
  6118.8 1564.88  6184.6 1566.24  6213.5 1567.41  6278.6 1568.01  6303.6 1568.59
#Mann=8,-1,0
  4498.2   0.035       0  4765.7    0.07       0  4997.1    0.07       0
  5001.8    0.07       0  5124.0   0.035       0  5622.9    0.07       0
  6184.6   0.035       0  6278.6    0.07       0
Bank Sta=4997.1,5001.8
Exp/Cntr=0.3,0.1

Type RM Length L Ch R = 1,24033,385,385,385
BEGIN DESCRIPTION:
Mapping XS f3305473
END DESCRIPTION:
XS GIS Cut Line= 3
      1614446.32      6984536.18      1614142.48      6984586.09
      1612925.06      6985050.49
#Sta/Elev= 30
  4701.9 1560.21  4741.3 1559.01  4774.2 1559.12  4794.4 1557.85  4838.0 1556.80
  4936.3 1555.88  4956.6 1554.84  4966.7 1553.40  4974.5 1552.94  4974.8 1552.44
  4978.9 1552.44  4979.3 1552.94  4986.3 1554.31  4991.4 1554.43  5084.0 1554.72
  5165.9 1554.89  5231.9 1556.51  5451.4 1556.61  5585.0 1555.98  5645.2 1557.16
  5705.4 1557.69  5745.6 1558.70  5899.9 1559.18  5954.7 1560.35  6023.9 1560.68
  6109.5 1562.95  6119.1 1562.60  6184.7 1563.42  6225.3 1564.68  6312.8 1565.63
#Mann=7,-1,0
  4701.9   0.035       0  4838.0    0.07       0  4974.5    0.07       0
  4979.3    0.07       0  5084.0   0.035       0  5451.4    0.07       0
  6225.3   0.035       0
Bank Sta=4974.5,4979.3
Exp/Cntr=0.3,0.1

Type RM Length L Ch R = 1,23648,161,161,161
BEGIN DESCRIPTION:
Mapping XS 5f2d4215
END DESCRIPTION:
XS GIS Cut Line= 3
      1614442.06      6984306.43      1614053.65      6984299.92
      1613048.33      6984826.41
#Sta/Elev= 30
  4614.5 1558.75  4641.6 1559.08  4691.6 1557.38  4794.9 1555.87  4891.6 1554.63
  4901.6 1554.31  4919.2 1552.21  4919.6 1551.71  4923.7 1551.71  4924.0 1552.21
  4941.6 1553.51  4961.6 1554.11  4971.6 1553.98  4981.6 1552.75  4991.6 1553.67
  5005.0 1553.61  5036.0 1554.94  5135.0 1555.17  5341.6 1555.31  5421.9 1555.34
  5565.1 1558.08  5659.0 1558.67  5703.2 1559.47  5890.5 1559.73  5949.7 1560.43
  6017.2 1560.27  6051.3 1560.71  6061.3 1561.52  6073.8 1560.96  6137.8 1561.78
#Mann=6,-1,0
  4614.5   0.035       0  4794.9    0.07       0  4919.2    0.07       0
  4924.0    0.07       0  5135.0   0.035       0  5341.6    0.07       0
Bank Sta=4919.2,4924
Exp/Cntr=0.3,0.1

Type RM Length L Ch R = 1,23487,151,151,151
BEGIN DESCRIPTION:
Mapping XS 7e564298
END DESCRIPTION:
XS GIS Cut Line= 3
      1614450.44      6984235.67      1614074.76      6984168.16
      1612454.50      6984304.59
#Sta/Elev= 30
  4618.3 1558.59  4685.6 1557.31  4735.6 1556.50  4755.9 1555.27  4831.3 1554.96
  4898.2 1553.43  4994.9 1552.91  4995.3 1552.41  4999.7 1552.91  5029.9 1554.52
  5160.4 1554.65  5592.3 1555.76  5852.8 1557.40  5895.0 1556.54  5933.1 1558.18
  5973.2 1558.22  5986.5 1561.39  6003.3 1565.80  6009.8 1566.00  6014.8 1560.74
  6033.4 1558.89  6093.6 1558.07  6113.7 1556.17  6163.9 1558.21  6204.0 1558.04
  6224.1 1556.64  6284.3 1558.27  6324.4 1558.05  6454.9 1562.39  6626.0 1565.11
#Mann=8,-1,0
  4618.3    0.07       0  4685.6   0.035       0  4831.3    0.07       0
  4994.9    0.07       0  4999.7    0.07       0  5160.4   0.035       0
  5592.3    0.07       0  5986.5   0.035       0
Bank Sta=4994.9,4999.7
Exp/Cntr=0.3,0.1

Type RM Length L Ch R = 1,23336,290,290,290
BEGIN DESCRIPTION:
Mapping XS b4b50856
END DESCRIPTION:
XS GIS Cut Line= 3
      1614452.64      6984170.99      1614146.67      6984040.79
      1612720.86      6983790.14
#Sta/Elev= 30
  4668.1 1557.96  4843.3 1554.24  5004.0 1553.47  5012.5 1551.97  5032.8 1553.50
  5063.2 1553.67  5101.1 1553.07  5114.0 1551.89  5125.9 1551.85  5142.0 1551.56
  5142.4 1551.06  5146.5 1551.06  5146.9 1551.56  5154.6 1551.92  5160.4 1553.15
  5165.5 1551.91  5185.1 1553.48  5225.7 1554.64  5378.0 1554.12  5551.1 1555.00
  5865.4 1556.59  5916.6 1555.40  5977.0 1555.21  6025.1 1556.00  6098.9 1555.32
  6138.7 1559.87  6210.6 1563.01  6291.8 1563.96  6376.1 1566.98  6448.3 1567.20
#Mann=5,-1,0
  4668.1    0.07       0  5125.9   0.035       0  5142.0    0.07       0
  5146.9   0.035       0  5551.1    0.07       0
Bank Sta=5142,5146.9
Exp/Cntr=0.3,0.1

Type RM Length L Ch R = 1,23046,134,134,134
BEGIN DESCRIPTION:
Mapping XS 3244a0ff
END DESCRIPTION:
XS GIS Cut Line= 4
      1614524.86      6984065.73      1613998.28      6983896.18
      1613479.96      6983537.49      1613324.86      6983251.35
#Sta/Elev= 30
  4446.8 1557.63  4459.1 1557.56  4467.7 1556.52  4478.2 1557.13  4499.2 1556.26
  4519.6 1556.62  4593.7 1554.96  4646.2 1555.12  4683.6 1553.19  4709.3 1552.72
  4811.9 1553.79  4919.8 1553.18  4983.0 1552.81  5145.0 1554.28  5237.6 1552.87
  5259.4 1553.93  5288.3 1553.16  5345.0 1553.53  5378.5 1552.50  5378.9 1552.00
  5383.4 1552.50  5395.7 1552.51  5404.5 1553.72  5446.4 1555.07  5453.9 1553.21
  5511.9 1554.40  5641.1 1554.81  5676.6 1556.36  5708.9 1559.88  5955.8 1564.82
#Mann=6,-1,0
  4446.8   0.035       0  4519.6    0.07       0  4919.8   0.035       0
  4983.0    0.07       0  5378.5    0.07       0  5383.4    0.07       0
Bank Sta=5378.5,5383.4
Exp/Cntr=0.3,0.1

Type RM Length L Ch R = 1,22912,348,348,348
BEGIN DESCRIPTION:
Mapping XS 27460a36
END DESCRIPTION:
XS GIS Cut Line= 3
      1614448.76      6984032.04      1614110.48      6983832.68
      1613762.48      6983257.51
#Sta/Elev= 30
  4607.8 1555.85  4744.7 1554.80  4809.5 1552.71  4877.5 1553.35  4957.5 1552.96
  4984.8 1551.55  5043.4 1552.64  5101.6 1552.12  5111.1 1551.49  5114.7 1550.57
  5115.0 1550.07  5119.2 1550.07  5119.6 1550.57  5154.0 1553.05  5175.3 1553.21
  5181.2 1554.22  5204.6 1555.56  5227.7 1555.44  5328.6 1551.07  5344.1 1552.13
  5349.9 1553.11  5365.4 1552.52  5386.8 1552.86  5408.1 1554.13  5423.6 1553.93
  5432.0 1554.47  5445.0 1554.48  5509.0 1557.31  5599.5 1559.59  5672.7 1561.69
#Mann=5,-1,0
  4607.8    0.07       0  5114.7    0.07       0  5119.6    0.07       0
  5432.0   0.035       0  5599.5    0.07       0
Bank Sta=5114.7,5119.6
Exp/Cntr=0.3,0.1

Type RM Length L Ch R = 1,22564,343,343,343
BEGIN DESCRIPTION:
Mapping XS e2e03882
END DESCRIPTION:
XS GIS Cut Line= 3
      1614294.64      6983753.57      1614163.11      6983534.79
      1613963.89      6983214.47
#Sta/Elev= 30
  4743.4 1554.28  4827.9 1553.29  4864.8 1553.38  4870.6 1552.87  4886.2 1553.68
  4892.0 1552.93  4901.6 1553.44  4907.5 1553.48  4913.4 1552.78  4923.1 1552.62
  4928.9 1551.84  4944.5 1551.32  4950.3 1550.59  4965.8 1548.02  4968.1 1547.97
  4968.6 1547.47  4974.7 1547.47  4975.2 1547.97  5023.9 1548.20  5075.9 1547.99
  5081.8 1548.91  5089.1 1551.14  5103.0 1551.63  5124.4 1551.98  5133.7 1552.73
  5176.2 1554.18  5249.4 1555.85  5309.2 1557.65  5310.6 1557.69  5375.9 1559.55
#Mann=5,-1,0
  4743.4    0.07       0  4968.1    0.07       0  4975.2    0.07       0
  5309.2   0.035       0  5310.6    0.07       0
Bank Sta=4968.1,4975.2
Exp/Cntr=0.3,0.1

Type RM Length L Ch R = 1,22221,152,152,152
BEGIN DESCRIPTION:
Mapping XS e427e591
END DESCRIPTION:
XS GIS Cut Line= 3
      1614428.65      6983998.49      1614418.24      6983373.50
      1614397.40      6982734.62
#Sta/Elev= 30
  4376.1 1555.32  4466.6 1554.08  4486.6 1554.26  4506.6 1553.37  4636.6 1552.21
  4726.6 1551.87  4796.6 1550.45  4816.7 1551.08  4846.7 1550.35  4856.7 1551.40
  4866.7 1551.76  4916.7 1551.89  4976.7 1550.95  4986.7 1550.31  4992.9 1549.30
  4993.4 1548.80  4999.5 1548.80  5000.0 1549.30  5016.7 1550.73  5036.7 1551.05
  5126.7 1551.40  5176.8 1551.17  5216.8 1551.55  5246.8 1551.10  5286.8 1551.94
  5326.9 1553.71  5346.9 1553.32  5376.9 1554.82  5456.9 1555.19  5640.4 1557.74
#Mann=3,-1,0
  4376.1    0.07       0  4992.9    0.07       0  5000.0    0.07       0
Bank Sta=4992.9,5000
Exp/Cntr=0.3,0.1

Type RM Length L Ch R = 1,22069,277,277,277
BEGIN DESCRIPTION:
Mapping XS 200cd539
END DESCRIPTION:
XS GIS Cut Line= 3
      1614544.97      6983955.10      1614525.87      6983267.60
      1614499.92      6982710.37
#Sta/Elev= 30
  4311.8 1556.30  4358.9 1555.65  4378.9 1555.78  4388.9 1555.00  4487.4 1552.90
  4529.0 1552.65  4569.0 1551.82  4619.0 1551.32  4649.0 1551.59  4709.1 1550.75
  4749.1 1551.30  4909.1 1551.08  4975.6 1549.82  4976.1 1549.32  4982.2 1549.32
  4982.7 1549.82  5009.2 1550.25  5049.2 1550.06  5079.3 1550.51  5139.3 1550.49
  5159.3 1550.97  5239.4 1551.15  5279.5 1551.84  5299.5 1551.55  5337.6 1551.69
  5342.6 1552.12  5429.6 1553.73  5529.7 1554.74  5549.8 1555.14  5557.4 1555.89
#Mann=3,-1,0
  4311.8   0.035       0  4975.6   0.035       0  4982.7   0.035       0
Bank Sta=4975.6,4982.7
Exp/Cntr=0.3,0.1

Type RM Length L Ch R = 1,21792,232,232,232
BEGIN DESCRIPTION:
Mapping XS 553d01d6
END DESCRIPTION:
XS GIS Cut Line= 3
      1614789.53      6984261.56      1614751.02      6983143.96
      1614730.00      6982462.95
#Sta/Elev= 30
  3878.6 1561.51  4172.3 1559.02  4295.8 1555.94  4332.4 1555.86  4432.5 1553.68
  4452.5 1552.05  4482.5 1550.95  4612.6 1550.47  4632.6 1549.88  4722.7 1550.51
  4752.7 1549.20  4792.7 1550.50  4964.9 1549.65  4999.2 1548.33  4999.7 1547.83
  5005.9 1547.83  5006.4 1548.33  5028.9 1549.86  5081.3 1550.43  5112.9 1551.16
  5122.9 1550.48  5182.9 1549.54  5212.9 1550.32  5323.0 1551.06  5393.0 1553.43
  5443.0 1554.05  5493.1 1556.04  5553.1 1557.15  5663.0 1557.64  5678.2 1557.57
#Mann=7,-1,0
  3878.6   0.035       0  4295.8    0.07       0  4964.9   0.035       0
  4999.2   0.035       0  5006.4   0.035       0  5081.3    0.07       0
  5663.0   0.035       0
Bank Sta=4999.2,5006.4
Exp/Cntr=0.3,0.1

Type RM Length L Ch R = 1,21560,534,534,534
BEGIN DESCRIPTION:
Mapping XS 908c9a8f
END DESCRIPTION:
XS GIS Cut Line= 3
      1615002.20      6984252.84      1614952.41      6983237.71
      1614930.00      6982412.97
#Sta/Elev= 30
  3977.4 1560.75  4052.3 1559.55  4242.6 1558.33  4372.7 1556.86  4415.0 1555.84
  4434.2 1556.22  4603.0 1554.17  4713.1 1551.43  4803.2 1550.10  4996.1 1549.53
  5019.9 1547.20  5020.4 1546.70  5026.6 1546.70  5027.1 1547.20  5043.5 1547.56
  5070.8 1549.65  5080.5 1550.48  5103.5 1550.44  5113.5 1551.74  5123.5 1550.24
  5133.5 1549.80  5243.6 1549.92  5273.6 1548.75  5313.3 1548.80  5343.6 1548.34
  5393.6 1549.62  5528.0 1551.32  5583.7 1553.45  5693.7 1555.95  5818.8 1556.50
#Mann=7,-1,0
  3977.4   0.035       0  4415.0    0.07       0  5019.9    0.07       0
  5027.1    0.07       0  5070.8   0.035       0  5313.3    0.07       0
  5528.0   0.035       0
Bank Sta=5019.9,5027.1
Exp/Cntr=0.3,0.1

Type RM Length L Ch R = 1,21026,119,119,119
BEGIN DESCRIPTION:
Mapping XS 90fdc292
END DESCRIPTION:
XS GIS Cut Line= 5
      1615278.00      6983829.93      1615294.42      6983409.59
      1615277.06      6983291.53      1615219.99      6983245.69
      1614991.63      6982631.78
#Sta/Elev= 30
  4455.8 1555.61  4647.9 1553.32  4748.0 1550.21  4831.3 1550.14  4910.2 1549.49
  4958.9 1545.37  4969.0 1543.97  4974.8 1542.08  5009.6 1541.96  5010.1 1541.46
  5017.4 1541.96  5049.7 1541.97  5063.1 1544.45  5069.0 1546.84  5095.4 1550.82
  5100.8 1552.82  5119.9 1554.31  5125.8 1554.07  5150.8 1549.75  5162.6 1549.16
  5258.6 1549.67  5297.2 1548.19  5327.5 1549.01  5382.9 1546.74  5418.6 1547.64
  5450.2 1547.30  5515.6 1548.83  5700.7 1551.56  5722.6 1553.06  5724.0 1553.18
#Mann=7,-1,0
  4455.8   0.035       0  4831.3    0.07       0  5009.6    0.07       0
  5017.4    0.07       0  5450.2   0.035       0  5515.6    0.07       0
  5722.6   0.035       0
Bank Sta=5009.6,5017.4
Exp/Cntr=0.3,0.1

Type RM Length L Ch R = 1,20907,41,41,41
BEGIN DESCRIPTION:
Mapping XS ce16e97c
END DESCRIPTION:
XS GIS Cut Line= 6
      1615347.45      6983812.49      1615344.77      6983385.28
      1615356.92      6983251.60      1615339.56      6983201.25
      1615240.82      6983165.83      1615023.51      6982584.64
#Sta/Elev= 30
  4386.7 1556.46  4631.2 1553.27  4743.1 1550.71  4841.3 1549.51  4869.1 1552.07
  4874.1 1550.91  4891.5 1553.82  4941.7 1552.56  4968.6 1553.13  4973.9 1551.53
  4994.3 1552.82  5016.9 1550.91  5024.0 1548.67  5029.3 1551.28  5054.8 1548.91
  5060.1 1551.40  5109.0 1554.24  5125.3 1550.02  5133.9 1549.10  5274.7 1548.91
  5310.4 1547.02  5356.3 1546.57  5356.8 1546.07  5364.1 1546.57  5420.8 1548.59
  5476.6 1549.10  5499.4 1549.18  5652.5 1551.12  5721.4 1553.39  5726.8 1553.40
#Mann=7,-1,0
  4386.7   0.035       0  4743.1    0.07       0  5356.3    0.07       0
  5364.1    0.07       0  5476.6   0.035       0  5499.4    0.07       0
  5721.4   0.035       0
Bank Sta=5356.3,5364.1
Exp/Cntr=0.3,0.1

Type RM Length L Ch R = 1,20866,195,195,195
BEGIN DESCRIPTION:
Mapping XS 04dbbb00
END DESCRIPTION:
XS GIS Cut Line= 6
      1615408.21      6983834.28      1615396.85      6983301.95
      1615396.85      6983199.52      1615369.07      6983173.48
      1615292.69      6983114.45      1615062.57      6982576.82
#Sta/Elev= 30
  4327.2 1558.02  4363.5 1557.82  4393.5 1556.60  4536.9 1554.45  4859.1 1549.01
  4923.6 1548.88  4960.3 1547.14  5016.9 1545.65  5017.4 1545.15  5024.2 1545.15
  5024.7 1545.65  5049.8 1547.10  5064.3 1547.12  5070.6 1548.46  5085.1 1548.82
  5129.9 1548.82  5147.2 1546.93  5153.5 1547.02  5158.9 1548.37  5169.0 1548.62
  5177.1 1547.31  5200.7 1547.32  5206.1 1548.32  5223.4 1548.88  5282.3 1546.61
  5321.3 1546.73  5382.1 1548.94  5495.3 1549.31  5625.8 1551.47  5681.5 1553.42
#Mann=4,-1,0
  4327.2   0.035       0  4536.9    0.07       0  5016.9    0.07       0
  5024.7    0.07       0
Bank Sta=5016.9,5024.7
Exp/Cntr=0.3,0.1

Type RM Length L Ch R = 1,20671,43,43,43
BEGIN DESCRIPTION:
Mapping XS fc65b836
END DESCRIPTION:
XS GIS Cut Line= 6
      1615493.55      6983449.39      1615530.01      6983241.01
      1615533.48      6983135.11      1615531.75      6983089.97
      1615491.82      6983032.68      1615084.59      6982552.26
#Sta/Elev= 30
  4635.0 1551.66  4731.6 1550.65  4809.0 1548.76  4829.3 1547.60  4899.6 1548.42
  4929.6 1544.72  4948.6 1543.31  4996.2 1543.52  5003.4 1542.61  5012.2 1542.91
  5014.3 1541.85  5014.8 1541.35  5022.2 1541.85  5024.5 1542.87  5054.1 1544.05
  5061.0 1545.82  5067.3 1548.55  5075.3 1548.49  5083.0 1549.88  5089.5 1549.27
  5097.3 1551.18  5111.6 1552.02  5132.4 1549.24  5146.7 1548.25  5210.4 1547.51
  5224.7 1546.46  5253.3 1545.87  5317.0 1547.84  5493.8 1549.34  5697.3 1553.63
#Mann=3,-1,0
  4635.0    0.07       0  5014.3    0.07       0  5022.2    0.07       0
Bank Sta=5014.3,5022.2
Exp/Cntr=0.3,0.1

Type RM Length L Ch R = 1,20628,36,36,36
BEGIN DESCRIPTION:
Mapping XS b80f5110
END DESCRIPTION:
XS GIS Cut Line= 6
      1615523.07      6983445.88      1615564.73      6983242.75
      1615575.15      6983116.01      1615569.94      6983074.34
      1615545.64      6983022.26      1615159.07      6982514.19
#Sta/Elev= 30
  4622.5 1551.57  4706.9 1551.01  4773.5 1549.63  4824.5 1547.44  4864.7 1548.38
  4892.0 1551.06  4897.0 1552.20  4975.2 1553.59  4994.4 1553.52  4998.8 1552.68
  5017.0 1553.87  5022.5 1552.33  5039.1 1553.16  5067.0 1552.99  5074.4 1552.33
  5081.5 1550.09  5084.7 1550.27  5110.6 1548.27  5136.7 1548.63  5160.5 1547.59
  5210.4 1547.44  5262.6 1545.74  5263.1 1545.24  5270.5 1545.74  5335.8 1547.67
  5413.4 1548.48  5489.0 1549.20  5538.9 1551.08  5629.4 1552.62  5694.9 1553.81
#Mann=8,-1,0
  4622.5    0.07       0  5084.7    0.16       0  5136.7    0.07       0
  5262.6    0.07       0  5270.5    0.07       0  5335.8   0.035       0
  5413.4    0.07       0  5629.4   0.035       0
Bank Sta=5262.6,5270.5
Exp/Cntr=0.3,0.1

Type RM Length L Ch R = 1,20592,250,250,250
BEGIN DESCRIPTION:
Mapping XS dc1855e6
END DESCRIPTION:
XS GIS Cut Line= 5
      1615542.18      6983477.08      1615604.66      6983223.65
      1615618.55      6983131.63      1615595.98      6983048.30
      1615211.53      6982433.41
#Sta/Elev= 30
  4558.8 1551.81  4592.7 1550.97  4640.2 1551.18  4774.1 1547.59  4858.2 1547.40
  4866.0 1548.07  4876.1 1547.41  4906.4 1548.21  4978.7 1546.81  4983.9 1549.21
  4996.8 1546.98  5008.0 1546.80  5013.9 1548.34  5029.2 1547.63  5035.1 1548.91
  5039.8 1548.54  5050.4 1548.67  5065.8 1547.47  5108.2 1548.30  5134.9 1547.59
  5217.9 1547.56  5256.4 1545.79  5256.9 1545.29  5264.3 1545.79  5372.7 1547.86
  5383.3 1547.75  5530.3 1551.05  5600.9 1551.89  5647.1 1553.62  5724.4 1554.09
#Mann=8,-1,0
  4558.8    0.07       0  5039.8    0.16       0  5134.9    0.07       0
  5256.4    0.07       0  5264.3    0.07       0  5372.7   0.035       0
  5383.3    0.07       0  5600.9   0.035       0
Bank Sta=5256.4,5264.3
Exp/Cntr=0.3,0.1

Type RM Length L Ch R = 1,20342,277,277,277
BEGIN DESCRIPTION:
Mapping XS 3bdf1856
END DESCRIPTION:
XS GIS Cut Line= 4
      1615878.96      6983322.93      1615809.53      6983031.29
      1615721.94      6982749.38      1615378.20      6982291.06
#Sta/Elev= 30
  4699.9 1553.29  4824.1 1551.27  4931.1 1548.84  4955.6 1547.44  4962.0 1545.62
  4972.2 1546.70  4982.5 1546.21  5021.6 1547.13  5063.1 1547.07  5068.4 1547.45
  5086.9 1546.52  5136.6 1546.69  5385.9 1547.13  5429.7 1545.94  5479.6 1545.61
  5490.3 1545.47  5490.8 1544.97  5497.7 1544.97  5498.2 1545.47  5500.5 1546.22
  5508.8 1545.85  5535.9 1546.51  5579.7 1546.68  5602.7 1547.92  5621.6 1548.97
  5679.7 1549.45  5729.7 1551.13  5811.0 1551.91  5820.3 1552.17  5867.8 1553.25
#Mann=9,-1,0
  4699.9    0.07       0  5021.6    0.16       0  5136.6    0.07       0
  5479.6   0.035       0  5490.3    0.07       0  5498.2   0.035       0
  5602.7    0.07       0  5811.0   0.035       0  5820.3    0.07       0
Bank Sta=5490.3,5498.2
Exp/Cntr=0.3,0.1

Type RM Length L Ch R = 1,20065,472,472,472
BEGIN DESCRIPTION:
Mapping XS 914a4f13
END DESCRIPTION:
XS GIS Cut Line= 4
      1616080.36      6983218.82      1616035.22      6982890.66
      1615977.93      6982661.50      1615518.51      6982247.20
#Sta/Elev= 30
  4665.6 1552.21  4741.9 1551.25  4868.3 1548.62  4885.9 1548.78  4898.6 1548.07
  4928.9 1547.83  4963.0 1546.69  4969.2 1546.28  4975.4 1545.24  4975.9 1544.74
  4982.8 1544.74  4983.3 1545.24  4995.7 1546.27  5016.7 1546.87  5021.9 1546.37
  5082.1 1545.26  5154.2 1546.29  5261.0 1546.21  5295.6 1546.29  5401.3 1546.23
  5450.3 1546.32  5471.2 1545.76  5556.4 1545.32  5605.7 1546.21  5619.9 1546.88
  5655.0 1547.04  5711.8 1549.15  5775.6 1549.56  5811.2 1550.93  5851.7 1550.97
#Mann=6,-1,0
  4665.6    0.07       0  4975.4    0.07       0  4983.3    0.07       0
  5261.0   0.035       0  5295.6    0.07       0  5401.3   0.035       0
Bank Sta=4975.4,4983.3
Exp/Cntr=0.3,0.1

Type RM Length L Ch R = 1,19593,277,277,277
BEGIN DESCRIPTION:
Mapping XS 92734ad7
END DESCRIPTION:
XS GIS Cut Line= 3
      1616400.84      6983114.62      1616236.77      6982502.61
      1615692.49      6982164.06
#Sta/Elev= 30
  4368.7 1552.52  4491.2 1550.86  4520.5 1551.12  4594.1 1549.37  4675.8 1546.28
  4680.9 1546.64  4686.1 1544.74  4696.5 1543.56  4737.9 1545.04  4775.2 1542.94
  4775.7 1542.44  4783.4 1542.94  4795.8 1543.33  4801.0 1544.64  4853.8 1545.34
  4882.9 1544.22  4903.6 1544.69  4915.8 1545.95  4945.0 1544.71  4973.0 1544.87
  5015.4 1544.18  5073.2 1545.23  5137.0 1545.70  5158.2 1545.10  5290.4 1546.42
  5441.5 1546.52  5514.7 1547.36  5522.6 1548.00  5589.5 1547.66  5643.3 1548.98
#Mann=8,-1,0
  4368.7    0.07       0  4594.1    0.16       0  4775.2   0.035       0
  4783.4    0.16       0  4853.8    0.07       0  4973.0   0.035       0
  5290.4    0.07       0  5589.5   0.035       0
Bank Sta=4775.2,4783.4
Exp/Cntr=0.3,0.1

Type RM Length L Ch R = 1,19316,375,375,375
BEGIN DESCRIPTION:
Mapping XS b5f83d01
END DESCRIPTION:
XS GIS Cut Line= 3
      1616682.07      6982828.12      1616450.31      6982338.55
      1615958.78      6982075.40
#Sta/Elev= 30
  4461.7 1552.21  4528.2 1550.65  4572.5 1547.04  4609.0 1545.06  4631.7 1544.56
  4716.3 1543.65  4908.6 1544.03  4978.5 1544.01  5003.4 1543.64  5005.3 1543.15
  5005.8 1542.65  5013.0 1542.65  5013.5 1543.15  5015.1 1543.52  5037.0 1543.53
  5089.4 1544.89  5236.2 1545.11  5250.7 1545.58  5258.9 1545.09  5281.6 1545.03
  5288.9 1545.66  5304.3 1545.25  5392.9 1545.45  5398.6 1545.96  5442.5 1545.92
  5496.9 1546.63  5508.5 1546.18  5518.9 1546.55  5546.5 1546.23  5560.9 1546.88
#Mann=5,-1,0
  4461.7    0.07       0  4908.6   0.035       0  5005.3   0.035       0
  5013.5   0.035       0  5089.4    0.07       0
Bank Sta=5005.3,5013.5
Exp/Cntr=0.3,0.1

Type RM Length L Ch R = 1,18941,583,583,583
BEGIN DESCRIPTION:
Mapping XS 483913aa
END DESCRIPTION:
XS GIS Cut Line= 3
      1616840.93      6982841.12      1616684.84      6982057.62
      1616048.05      6981991.60
#Sta/Elev= 30
  4201.1 1549.50  4207.6 1549.84  4253.6 1548.62  4258.7 1549.08  4304.7 1547.43
  4309.8 1547.81  4355.8 1546.06  4377.6 1546.15  4406.8 1545.02  4482.6 1543.90
  4500.0 1543.13  4523.6 1542.83  4565.2 1542.39  4601.9 1543.88  4662.3 1544.43
  4722.9 1543.71  4769.5 1543.31  4871.7 1543.87  4897.6 1543.28  5034.8 1542.53
  5080.3 1543.08  5106.3 1542.28  5106.8 1541.78  5114.0 1541.78  5114.5 1542.28
  5311.5 1544.74  5473.4 1544.93  5492.5 1544.73  5512.6 1545.32  5640.2 1546.11
#Mann=8,-1,0
  4201.1   0.035       0  4482.6    0.07       0  4523.6   0.035       0
  4722.9    0.07       0  5034.8   0.035       0  5106.3    0.07       0
  5114.5   0.035       0  5473.4    0.07       0
Bank Sta=5106.3,5114.5
Exp/Cntr=0.3,0.1

Type RM Length L Ch R = 1,18358,869,869,869
BEGIN DESCRIPTION:
Mapping XS d8b441be
END DESCRIPTION:
XS GIS Cut Line= 3
      1617142.98      6983264.06      1617182.04      6982261.47
      1617242.80      6981076.58
#Sta/Elev= 30
  3999.6 1553.56  4112.5 1552.66  4126.2 1552.32  4180.4 1551.21  4257.6 1548.63
  4375.9 1545.94  4456.0 1542.95  4636.6 1541.99  4746.2 1541.73  4756.2 1542.21
  4859.4 1542.53  4926.4 1541.65  4966.4 1542.07  4995.8 1541.58  4996.3 1541.08
  5008.1 1541.08  5008.6 1541.58  5076.5 1541.91  5208.8 1543.97  5246.7 1545.23
  5366.9 1546.79  5520.5 1547.61  5544.3 1547.68  5617.2 1548.00  5684.5 1549.12
  5737.4 1549.45  5743.3 1549.00  5950.1 1551.27  5967.6 1551.42  6189.4 1553.94
#Mann=14,-1,0
  3999.6   0.035       0  4112.5    0.07       0  4126.2   0.035       0
  4257.6    0.07       0  4636.6   0.035       0  4859.4    0.07       0
  4995.8    0.07       0  5008.6    0.07       0  5208.8   0.035       0
  5520.5    0.07       0  5544.3   0.035       0  5684.5    0.07       0
  5950.1   0.035       0  5967.6    0.07       0
Bank Sta=4995.8,5008.6
Exp/Cntr=0.3,0.1

Type RM Length L Ch R = 1,17489,918,918,918
BEGIN DESCRIPTION:
Mapping XS 95796bdd
END DESCRIPTION:
XS GIS Cut Line= 3
      1617932.90      6983203.27      1617807.04      6982634.73
      1617702.87      6981363.00
#Sta/Elev= 30
  4415.7 1558.88  4563.6 1555.86  4617.5 1555.39  4718.1 1552.60  4753.5 1552.11
  4912.7 1547.14  4963.9 1543.67  4993.8 1539.84  5024.8 1539.35  5028.2 1537.69
  5028.7 1537.19  5041.0 1537.19  5041.5 1537.69  5044.9 1538.63  5054.9 1539.36
  5087.1 1540.61  5155.3 1540.48  5239.0 1541.82  5240.1 1541.85  5243.6 1541.93
  5275.7 1542.90  5476.3 1545.92  5633.8 1547.26  5732.3 1548.15  5817.3 1548.90
  5998.1 1550.20  6018.1 1551.32  6038.2 1550.80  6168.6 1551.78  6274.0 1553.49
#Mann=9,-1,0
  4415.7   0.035       0  5028.2   0.035       0  5041.5   0.035       0
  5239.0    0.07       0  5240.1   0.035       0  5243.6    0.07       0
  5633.8   0.035       0  5732.3    0.07       0  5817.3   0.035       0
Bank Sta=5028.2,5041.5
Exp/Cntr=0.3,0.1

Type RM Length L Ch R = 1,16571,550,550,550
BEGIN DESCRIPTION:
Mapping XS a38c1cdf
END DESCRIPTION:
XS GIS Cut Line= 3
      1619169.91      6982613.05      1618406.00      6982027.09
      1618015.35      6981276.19
#Sta/Elev= 30
  4044.5 1556.77  4158.7 1554.86  4201.9 1555.00  4223.1 1553.99  4351.8 1551.83
  4365.8 1552.36  4393.6 1550.73  4408.0 1550.09  4416.2 1551.12  4443.3 1551.03
  4529.6 1548.88  4592.9 1548.56  4715.3 1543.76  4794.2 1539.48  4979.1 1538.72
  4985.4 1538.28  4993.1 1534.24  4993.6 1533.74  5006.6 1534.24  5007.3 1536.69
  5021.7 1539.09  5046.7 1539.24  5082.4 1539.01  5133.8 1540.16  5252.0 1544.29
  5400.8 1548.31  5423.3 1550.25  5430.4 1549.93  5496.8 1552.31  5853.7 1557.31
#Mann=7,-1,0
  4044.5   0.045       0  4393.6    0.07       0  4993.1    0.07       0
  5006.6    0.07       0  5046.7   0.035       0  5133.8    0.07       0
  5252.0   0.035       0
Bank Sta=4993.1,5006.6
Exp/Cntr=0.3,0.1

Type RM Length L Ch R = 1,16021,238,238,238
BEGIN DESCRIPTION:
Mapping XS f79eea15
END DESCRIPTION:
XS GIS Cut Line= 3
      1619212.88      6981885.18      1618804.00      6981682.04
      1618236.75      6981382.80
#Sta/Elev= 30
  4542.8 1547.69  4732.8 1545.48  4748.5 1546.02  4798.9 1542.39  4842.9 1541.63
  4882.9 1541.56  4888.5 1542.30  4942.4 1541.31  4978.1 1539.57  4987.1 1538.95
  4998.3 1535.99  5001.6 1535.99  5002.7 1533.03  5003.2 1532.53  5016.3 1533.03
  5017.0 1534.95  5022.6 1535.88  5039.0 1537.46  5061.0 1538.23  5088.7 1537.58
  5105.1 1535.37  5111.3 1537.20  5121.4 1537.87  5215.2 1538.45  5291.9 1540.88
  5336.0 1540.93  5495.8 1550.34  5556.3 1553.07  5626.3 1554.64  5640.7 1555.03
#Mann=7,-1,0
  4542.8   0.045       0  4732.8    0.07       0  4842.9   0.035       0
  5002.7   0.035       0  5016.3   0.035       0  5556.3    0.07       0
  5626.3   0.035       0
Bank Sta=5002.7,5016.3
Exp/Cntr=0.3,0.1

Type RM Length L Ch R = 1,15783,728,728,728
BEGIN DESCRIPTION:
Mapping XS ed98349a
END DESCRIPTION:
XS GIS Cut Line= 3
      1619163.34      6981572.66      1618754.52      6981460.69
      1618328.76      6981278.96
#Sta/Elev= 30
  4576.4 1542.16  4601.5 1542.01  4719.8 1540.37  4731.0 1537.84  4740.6 1537.00
  4771.7 1538.53  4792.4 1535.11  4823.5 1536.50  4906.5 1536.36  4913.7 1538.41
  4918.9 1538.11  4927.2 1541.27  4937.6 1541.23  4947.9 1539.13  4953.4 1536.43
  5010.6 1536.18  5016.6 1533.50  5017.1 1533.00  5030.2 1533.50  5032.4 1535.04
  5041.6 1536.54  5047.0 1535.43  5070.6 1538.02  5117.8 1540.79  5123.3 1539.46
  5206.3 1541.59  5282.5 1547.01  5383.4 1551.85  5434.7 1554.82  5463.2 1554.96
#Mann=5,-1,0
  4576.4    0.07       0  4601.5   0.035       0  5016.6   0.035       0
  5030.2   0.035       0  5383.4    0.07       0
Bank Sta=5016.6,5030.2
Exp/Cntr=0.3,0.1

Type RM Length L Ch R = 1,15055,494,494,494
BEGIN DESCRIPTION:
Mapping XS 98c083b2
END DESCRIPTION:
XS GIS Cut Line= 3
      1619282.22      6981521.76      1619248.37      6981037.44
      1619061.20      6980712.49
#Sta/Elev= 30
  4515.3 1541.97  4550.7 1541.68  4599.3 1539.40  4639.4 1538.82  4649.4 1538.06
  4679.5 1538.00  4687.5 1537.44  4834.4 1535.34  4930.1 1535.30  4970.2 1536.28
  4976.3 1535.34  4981.3 1537.20  4990.2 1534.31  4999.1 1532.31  5003.4 1532.31
  5004.8 1531.39  5005.3 1530.89  5018.0 1530.89  5018.5 1531.39  5033.3 1534.94
  5039.1 1535.11  5046.3 1536.27  5054.9 1539.27  5060.6 1539.80  5076.4 1543.59
  5100.0 1545.29  5141.1 1547.01  5172.7 1546.68  5336.8 1549.50  5375.8 1549.31
#Mann=6,-1,0
  4515.3    0.07       0  4999.1    0.16       0  5004.8    0.07       0
  5018.5    0.16       0  5100.0    0.07       0  5336.8   0.035       0
Bank Sta=5004.8,5018.5
Exp/Cntr=0.3,0.1

Type RM Length L Ch R = 1,14561,533,533,533
BEGIN DESCRIPTION:
Mapping XS b01346a4
END DESCRIPTION:
XS GIS Cut Line= 3
      1619774.41      6981670.20      1619691.08      6981092.12
      1619462.30      6980501.97
#Sta/Elev= 30
  4411.3 1548.71  4423.6 1548.46  4440.5 1547.02  4534.8 1544.26  4544.9 1543.06
  4565.1 1543.26  4676.2 1540.14  4722.1 1539.89  4736.8 1538.69  4787.4 1537.36
  4817.7 1535.75  4878.3 1534.32  4994.6 1533.34  4995.1 1532.84  5008.3 1532.84
  5008.8 1533.34  5010.5 1534.32  5056.2 1534.21  5086.1 1533.39  5140.6 1534.25
  5244.2 1534.69  5428.8 1537.18  5450.2 1537.91  5461.0 1538.90  5472.9 1541.16
  5482.4 1541.63  5497.4 1543.35  5503.9 1544.81  5514.6 1545.59  5628.3 1548.57
#Mann=3,-1,0
  4411.3    0.07       0  4994.6    0.07       0  5008.8    0.07       0
Bank Sta=4994.6,5008.8
Exp/Cntr=0.3,0.1

Type RM Length L Ch R = 1,14028,686,686,686
BEGIN DESCRIPTION:
Mapping XS c062f7dc
END DESCRIPTION:
XS GIS Cut Line= 3
      1620503.62      6981256.22      1620125.98      6980917.64
      1619572.65      6980431.86
#Sta/Elev= 30
  4492.8 1544.29  4517.2 1543.72  4733.5 1538.62  4765.4 1537.78  4809.4 1536.74
  4852.0 1536.47  4872.9 1537.06  4890.5 1535.86  4895.1 1535.25  4922.3 1535.04
  4929.7 1534.53  4936.5 1533.10  4957.8 1532.41  4958.3 1531.91  4971.5 1531.91
  4972.0 1532.41  4972.4 1532.90  5007.5 1533.97  5142.2 1533.11  5347.3 1534.68
  5418.4 1536.15  5432.6 1535.47  5475.3 1536.08  5560.2 1538.42  5567.3 1539.19
  5574.0 1539.02  5624.3 1541.21  5652.7 1544.64  5689.3 1547.84  5736.3 1549.48
#Mann=9,-1,0
  4492.8   0.035       0  4517.2    0.07       0  4733.5   0.035       0
  4765.4    0.07       0  4890.5   0.035       0  4895.1    0.07       0
  4957.8    0.07       0  4972.0    0.07       0  5689.3   0.035       0
Bank Sta=4957.8,4972
Exp/Cntr=0.3,0.1

Type RM Length L Ch R = 1,13342,439,439,439
BEGIN DESCRIPTION:
Mapping XS fa334204
END DESCRIPTION:
XS GIS Cut Line= 3
      1621492.53      6981009.46      1620352.89      6980367.25
      1619574.11      6980145.74
#Sta/Elev= 30
  3694.4 1544.20  3848.3 1543.76  4207.4 1537.37  4382.9 1535.78  4501.4 1536.84
  4517.3 1536.69  4523.0 1535.44  4632.8 1534.61  4655.8 1533.38  4911.7 1533.40
  4949.0 1532.38  4970.9 1531.50  4977.1 1529.49  4991.3 1528.57  4991.8 1528.07
  5005.6 1528.57  5017.0 1531.02  5031.5 1532.14  5078.2 1530.98  5177.1 1533.06
  5196.8 1531.63  5208.3 1532.99  5291.4 1533.19  5395.4 1535.24  5532.8 1539.46
  5621.7 1543.47  5639.6 1544.68  5665.7 1548.34  5688.8 1549.20  5812.2 1555.84
#Mann=8,-1,0
  3694.4   0.045       0  4207.4   0.035       0  4949.0    0.16       0
  4991.3    0.07       0  5005.6    0.16       0  5078.2   0.035       0
  5621.7    0.07       0  5688.8   0.035       0
Bank Sta=4991.3,5005.6
Exp/Cntr=0.3,0.1

Type RM Length L Ch R = 1,12903,305,305,305
BEGIN DESCRIPTION:
Mapping XS b4e40384
END DESCRIPTION:
XS GIS Cut Line= 3
      1621436.09      6980827.17      1620407.14      6979946.25
      1620220.96      6979712.45
#Sta/Elev= 30
  3646.4 1542.24  3725.0 1541.73  3772.2 1539.82  3866.6 1538.70  3909.4 1536.85
  4001.6 1536.66  4008.2 1534.49  4100.4 1531.89  4327.6 1531.59  4362.7 1530.75
  4511.2 1531.79  4554.8 1531.13  4596.5 1532.18  4658.8 1531.93  4887.7 1531.52
  4958.7 1531.28  4970.0 1530.22  4986.6 1528.31  4987.1 1527.81  5001.1 1528.31
  5023.2 1529.99  5029.5 1531.34  5050.4 1532.13  5079.2 1538.51  5087.2 1542.69
  5093.6 1542.77  5101.0 1547.19  5136.9 1555.87  5186.5 1557.44  5299.8 1557.10
#Mann=8,-1,0
  3646.4   0.045       0  3772.2   0.035       0  4511.2    0.07       0
  4658.8   0.035       0  4887.7    0.16       0  4970.0    0.07       0
  4986.6    0.07       0  5001.1    0.07       0
Bank Sta=4986.6,5001.1
Exp/Cntr=0.3,0.1

Type RM Length L Ch R = 1,12598,374,374,374
BEGIN DESCRIPTION:
Mapping XS a88d0811
END DESCRIPTION:
XS GIS Cut Line= 3
      1621318.87      6980662.20      1620660.06      6979793.30
      1620514.22      6979565.85
#Sta/Elev= 30
  3906.9 1539.15  3956.9 1537.96  3990.8 1537.34  4005.3 1535.86  4019.3 1536.48
  4034.4 1536.87  4140.5 1532.16  4225.9 1530.82  4419.3 1529.96  4622.5 1530.73
  4701.3 1530.42  4723.4 1530.69  4783.3 1530.82  4833.2 1529.88  4847.8 1530.77
  4912.3 1530.64  4933.1 1530.40  4940.4 1528.53  4940.9 1528.03  4954.9 1528.53
  5025.8 1531.76  5039.8 1534.62  5055.0 1539.35  5063.0 1542.94  5070.2 1547.81
  5091.4 1556.86  5098.6 1559.00  5193.7 1561.59  5200.4 1561.01  5267.5 1562.22
#Mann=9,-1,0
  3906.9   0.035       0  3956.9    0.07       0  4019.3   0.035       0
  4622.5    0.07       0  4701.3   0.035       0  4723.4    0.16       0
  4940.4    0.07       0  4954.9    0.16       0  5025.8    0.07       0
Bank Sta=4940.4,4954.9
Exp/Cntr=0.3,0.1

Type RM Length L Ch R = 1,12224,58,58,58
BEGIN DESCRIPTION:
Mapping XS 4459c630
END DESCRIPTION:
XS GIS Cut Line= 4
      1621410.02      6980718.61      1621002.08      6979880.98
      1621002.08      6979697.81      1620953.52      6979482.78
#Sta/Elev= 30
  3882.2 1540.82  3924.9 1539.56  3983.0 1539.59  3993.0 1538.89  4020.6 1538.51
  4027.5 1537.48  4043.1 1537.30  4060.1 1538.20  4087.8 1536.88  4161.4 1535.53
  4216.6 1532.61  4246.0 1531.82  4593.8 1528.27  4620.9 1527.55  4621.4 1527.05
  4635.4 1527.55  4650.4 1528.69  4725.0 1529.93  4836.9 1529.95  4856.9 1529.48
  4866.9 1527.64  4886.9 1529.77  4926.9 1530.76  4954.9 1528.71  5004.2 1528.58
  5047.4 1533.58  5054.5 1533.65  5095.8 1535.12  5150.6 1534.54  5217.5 1536.70
#Mann=8,-1,0
  3882.2   0.035       0  3993.0    0.07       0  4087.8   0.035       0
  4593.8    0.16       0  4620.9    0.07       0  4635.4    0.16       0
  4954.9    0.07       0  5054.5   0.035       0
Bank Sta=4620.9,4635.4
Exp/Cntr=0.3,0.1

Type RM Length L Ch R = 1,12166,993,993,993
BEGIN DESCRIPTION:
Mapping XS 7ddd46a1
END DESCRIPTION:
XS GIS Cut Line= 4
      1621531.57      6980883.60      1621079.73      6979793.41
      1621057.63      6979680.45      1621005.55      6979444.35
#Sta/Elev= 30
  3705.8 1543.29  3722.7 1543.84  3761.4 1542.39  3861.3 1541.50  3995.1 1539.65
  4027.3 1538.31  4058.3 1538.83  4117.5 1537.14  4199.0 1536.05  4306.2 1531.78
  4471.2 1529.29  4534.6 1526.42  4548.2 1524.21  4564.8 1524.13  4565.3 1523.63
  4579.4 1524.13  4610.3 1527.95  4642.8 1529.33  4784.8 1529.23  4808.7 1528.18
  4816.0 1529.24  4834.9 1529.09  4938.5 1530.16  4993.6 1528.68  5013.8 1526.28
  5038.9 1531.86  5054.7 1534.12  5103.0 1535.94  5240.6 1539.89  5242.8 1539.89
#Mann=11,-1,0
  3705.8   0.045       0  3861.3   0.035       0  3995.1    0.07       0
  4117.5   0.035       0  4564.8   0.035       0  4579.4   0.035       0
  4834.9    0.07       0  4938.5   0.035       0  5038.9    0.07       0
  5103.0   0.035       0  5240.6    0.07       0
Bank Sta=4564.8,4579.4
Exp/Cntr=0.3,0.1

Type RM Length L Ch R = 1,11173,750,750,750
BEGIN DESCRIPTION:
Mapping XS f630e44b
END DESCRIPTION:
XS GIS Cut Line= 3
      1621708.84      6980582.81      1621441.27      6979851.21
      1621076.85      6979207.73
#Sta/Elev= 30
  4221.0 1541.05  4457.8 1538.16  4655.8 1534.20  4662.7 1533.39  4681.0 1533.31
  4736.8 1531.28  4747.9 1531.49  4767.3 1530.34  4811.8 1529.12  4896.4 1528.16
  4970.4 1527.30  4992.8 1524.97  4998.7 1522.96  4999.2 1522.46  5012.9 1522.46
  5013.4 1522.96  5037.8 1525.31  5049.7 1528.28  5059.4 1528.90  5115.9 1529.14
  5224.4 1529.27  5344.4 1529.96  5404.3 1531.56  5447.6 1534.78  5463.4 1534.72
  5485.1 1535.53  5490.9 1536.34  5506.7 1536.19  5571.7 1538.29  5739.5 1541.93
#Mann=8,-1,0
  4221.0    0.07       0  4457.8   0.035       0  4896.4    0.16       0
  4998.7    0.07       0  5013.4    0.16       0  5115.9   0.035       0
  5224.4    0.16       0  5344.4   0.035       0
Bank Sta=4998.7,5013.4
Exp/Cntr=0.3,0.1

Type RM Length L Ch R = 1,10423,421,421,421
BEGIN DESCRIPTION:
Mapping XS 2361f0fc
END DESCRIPTION:
XS GIS Cut Line= 4
      1621728.41      6980221.66      1621750.98      6979436.99
      1621636.97      6979356.14      1621413.00      6979078.35
#Sta/Elev= 30
  4074.7 1535.55  4158.4 1533.44  4168.4 1533.71  4188.4 1532.62  4288.5 1529.91
  4408.5 1529.28  4536.6 1527.26  4578.6 1526.77  4598.6 1527.53  4608.6 1526.99
  4764.5 1527.27  4838.7 1526.32  4914.2 1526.87  4985.6 1526.12  4997.6 1523.67
  5000.7 1523.67  5006.1 1523.15  5006.6 1522.65  5020.3 1522.65  5020.8 1523.15
  5027.8 1526.47  5035.6 1528.04  5048.7 1529.04  5071.0 1529.06  5091.8 1530.09
  5120.6 1530.21  5215.2 1532.63  5219.8 1533.26  5291.7 1534.60  5356.3 1537.20
#Mann=7,-1,0
  4074.7   0.035       0  4536.6    0.07       0  4764.5    0.16       0
  5000.7    0.07       0  5006.1    0.07       0  5020.8    0.07       0
  5215.2   0.035       0
Bank Sta=5006.1,5020.8
Exp/Cntr=0.3,0.1

Type RM Length L Ch R = 1,10002,326,326,326
BEGIN DESCRIPTION:
Mapping XS d4d1a4b5
END DESCRIPTION:
XS GIS Cut Line= 4
      1621771.81      6980223.47      1621840.45      6979759.66
      1621940.79      6979422.12      1622274.21      6978601.57
#Sta/Elev= 30
  4180.5 1536.43  4226.5 1535.05  4246.7 1533.93  4303.5 1533.00  4357.9 1530.91
  4428.6 1529.84  4499.4 1529.50  4617.3 1527.67  4651.4 1527.19  4757.9 1526.10
  4894.8 1525.23  4911.9 1525.73  4922.3 1527.24  4928.0 1527.35  4943.2 1523.88
  4958.9 1522.45  4959.4 1521.95  4973.5 1521.95  4974.0 1522.45  4994.4 1523.48
  4999.7 1526.31  5016.7 1528.08  5022.7 1527.93  5107.1 1527.72  5362.1 1529.19
  5393.5 1528.85  5423.0 1529.46  5491.7 1529.63  5599.6 1532.26  5887.2 1534.62
#Mann=7,-1,0
  4180.5   0.035       0  4617.3    0.07       0  4651.4   0.035       0
  4757.9    0.07       0  4958.9    0.07       0  4974.0    0.07       0
  5022.7    0.07       0
Bank Sta=4958.9,4974
Exp/Cntr=0.3,0.1

Type RM Length L Ch R = 1,9676,443,443,443
BEGIN DESCRIPTION:
Mapping XS 54649a0e
END DESCRIPTION:
XS GIS Cut Line= 4
      1621768.34      6980351.93      1621877.71      6979938.72
      1622225.09      6979438.93      1622545.62      6978745.97
#Sta/Elev= 30
  3962.2 1538.14  3983.8 1537.81  4235.2 1532.60  4281.6 1531.15  4321.8 1530.94
  4356.8 1529.65  4414.1 1528.86  4445.8 1528.98  4481.6 1528.18  4618.6 1527.08
  4740.8 1525.19  4827.3 1524.48  4869.1 1524.89  4884.0 1526.37  4926.4 1526.23
  4955.6 1526.86  4962.9 1526.25  4970.4 1522.97  4983.8 1522.60  4984.3 1522.10
  4998.5 1522.10  4999.0 1522.60  5012.9 1523.02  5030.3 1526.01  5035.8 1525.65
  5058.8 1527.21  5173.4 1527.92  5270.6 1529.65  5436.6 1531.18  5761.8 1533.29
#Mann=5,-1,0
  3962.2    0.07       0  3983.8   0.035       0  4414.1    0.07       0
  4983.8    0.07       0  4999.0    0.07       0
Bank Sta=4983.8,4999
Exp/Cntr=0.3,0.1

Type RM Length L Ch R = 1,9233,193,193,193
BEGIN DESCRIPTION:
Mapping XS dc2dfc68
END DESCRIPTION:
XS GIS Cut Line= 3
      1621927.61      6979909.14      1622303.22      6979756.64
      1623071.73      6979420.73
#Sta/Elev= 30
  4592.5 1528.65  4714.5 1528.00  4845.7 1525.56  4904.6 1525.15  4952.8 1523.97
  4967.4 1524.57  4976.9 1523.39  4982.3 1523.79  4989.0 1522.78  4998.5 1522.49
  4999.0 1521.99  5013.2 1521.99  5013.7 1522.49  5105.2 1524.41  5110.6 1524.09
  5119.9 1524.60  5128.6 1525.79  5174.4 1525.46  5233.1 1526.04  5326.7 1525.85
  5605.5 1528.23  5621.9 1528.70  5634.7 1528.39  5658.1 1528.81  5665.6 1527.76
  5681.5 1529.38  5687.4 1529.52  5720.1 1529.15  5780.5 1529.43  5836.6 1529.46
#Mann=5,-1,0
  4592.5    0.07       0  4998.5    0.07       0  5013.7    0.07       0
  5605.5   0.035       0  5780.5    0.07       0
Bank Sta=4998.5,5013.7
Exp/Cntr=0.3,0.1

Type RM Length L Ch R = 1,9040,93,93,93
BEGIN DESCRIPTION:
Mapping XS 3a311335
END DESCRIPTION:
XS GIS Cut Line= 3
      1621942.50      6979955.86      1622303.22      6979949.34
      1622888.77      6979666.17
#Sta/Elev= 30
  4637.8 1529.30  4690.3 1529.00  4795.7 1526.83  4920.3 1524.90  4930.3 1525.09
  4950.3 1524.48  4970.4 1524.28  4980.4 1522.99  4982.8 1521.38  4983.3 1520.88
  4997.5 1520.88  4998.0 1521.38  5002.3 1521.70  5015.2 1521.43  5022.8 1522.58
  5037.8 1523.17  5060.4 1523.14  5067.2 1523.63  5083.0 1523.82  5105.6 1524.60
  5111.6 1524.19  5122.6 1524.14  5300.5 1524.98  5314.4 1525.33  5322.7 1525.07
  5444.4 1525.38  5600.4 1527.02  5608.1 1527.38  5623.0 1527.28  5649.0 1527.73
#Mann=4,-1,0
  4637.8    0.07       0  4982.8    0.07       0  4998.0    0.07       0
  5623.0   0.035       0
Bank Sta=4982.8,4998
Exp/Cntr=0.3,0.1

Type RM Length L Ch R = 1,8947,404,404,404
BEGIN DESCRIPTION:
Mapping XS d4b30d5b
END DESCRIPTION:
XS GIS Cut Line= 3
      1621992.03      6980063.93      1622347.49      6980027.47
      1622881.13      6979701.59
#Sta/Elev= 30
  4645.9 1530.42  4679.0 1529.61  4739.4 1529.47  4753.7 1528.79  4829.8 1527.46
  4860.0 1526.42  4940.4 1525.15  4970.6 1523.78  4983.0 1520.60  4983.5 1520.10
  4997.9 1520.10  4998.4 1520.60  4999.5 1522.13  5003.2 1522.13  5009.0 1522.97
  5014.8 1522.62  5023.7 1522.64  5030.3 1523.15  5036.2 1522.77  5045.8 1522.94
  5058.9 1524.35  5072.9 1525.12  5094.2 1524.17  5117.5 1524.27  5140.6 1523.84
  5220.0 1524.84  5283.9 1525.15  5467.7 1525.31  5611.3 1527.07  5628.5 1527.61
#Mann=4,-1,0
  4645.9    0.07       0  4983.0    0.07       0  4998.4    0.07       0
  5611.3   0.035       0
Bank Sta=4983,4998.4
Exp/Cntr=0.3,0.1
