--- Swager Creek.prj (project) ---

Proj Title=Swager Creek Base Level Engineering
Current Plan=p01
Default Exp/Contr=0.3,0.1
English Units
Geom File=g01
Flow File=f01
Plan File=p01
BEGIN DESCRIPTION:
Swager Creek
END DESCRIPTION:

--- Swager Creek.p01 (plan) ---

Plan Title=Multiple Run
Short Identifier=Multiple
Geom File=g01
Flow File=f01
Subcritical Flow
K Sum by GR= 0
Std Step Tol= 0.01
Critical Tol= 0.01
Num of Std Step Trials= 20
Max Error Tol= 0.3
Flow Tol Ratio= 0.001
Split Flow NTrial= 30
Split Flow Tol= 0.02
Split Flow Ratio= 0.02
Log Output Level= 0
Friction Slope Method= 1
Unsteady Friction Slope Method= 2
Unsteady Bridges Friction Slope Method= 1
Parabolic Critical Depth
Global Vel Dist=  1 , 1 , 1
Global Log Level= 0
CheckData=True
Encroach Param= -1, 0, 0, 0
BEGIN DESCRIPTION:
Multiple Run
END DESCRIPTION:

--- Swager Creek.f01 (steady flow) ---

Flow Title=Multiple
Number of Profiles=7
Profile Names=10-year,25-year,50-year,1pct_min,100-year,1pct_plu,500-year
River Rch & RM= Swager Creek,Reach-1,67896
     262     361     441     269     537    1072     804
River Rch & RM= Swager Creek,Reach-1,64486
     349     486     600     369     736    1468    1119
River Rch & RM= Swager Creek,Reach-1,61614
     456     644     801     496     989    1973    1525
River Rch & RM= Swager Creek,Reach-1,53291
     488     691     862     534    1066    2128    1653
River Rch & RM= Swager Creek,Reach-1,51786
     534     762     955     595    1187    2368    1856
River Rch & RM= Swager Creek,Reach-1,47310
    1150    1699    2180    1386    2766    5519    4516
River Rch & RM= Swager Creek,Reach-1,35274
    1436    2136    2755    1760    3512    7008    5787
River Rch & RM= Swager Creek,Reach-1,28698
    1501    2236    2887    1846    3683    7349    6079
River Rch & RM= Swager Creek,Reach-1,25076
    1572    2344    3027    1937    3864    7710    6381
River Rch & RM= Swager Creek,Reach-1,17460
    1800    2698    3499    2247    4483    8944    7456
River Rch & RM= Swager Creek,Reach-1,6577
    1831    2746    3561    2286    4562    9103    7589
River Rch & RM= Swager Creek,Reach-1,1434
    2171    3275    4265    2749    5484   10943    9192
Boundary for River Rch & Prof#=Swager Creek,Reach-1,1
Up Type=0
Dn Type=3
Dn Slope=0.005
Boundary for River Rch & Prof#=Swager Creek,Reach-1,2
Up Type=0
Dn Type=3
Dn Slope=0.005
Boundary for River Rch & Prof#=Swager Creek,Reach-1,3
Up Type=0
Dn Type=3
Dn Slope=0.005
Boundary for River Rch & Prof#=Swager Creek,Reach-1,4
Up Type=0
Dn Type=3
Dn Slope=0.005
Boundary for River Rch & Prof#=Swager Creek,Reach-1,5
Up Type=0
Dn Type=3
Dn Slope=0.005
Boundary for River Rch & Prof#=Swager Creek,Reach-1,6
Up Type=0
Dn Type=3
Dn Slope=0.005
Boundary for River Rch & Prof#=Swager Creek,Reach-1,7
Up Type=0
Dn Type=3
Dn Slope=0.005

--- Swager Creek.g01 (geometry) ---

Geom Title=Existing Conditions

River Reach=Swager Creek,Reach-1
Reach XY= 30
      1682105.00      6971538.00      1681449.93      6973835.93
      1679912.95      6973385.19      1679791.03      6972788.55
      1676875.36      6973338.36      1675801.77      6972945.83
      1673145.34      6974336.63      1670906.50      6973841.46
      1669107.43      6975482.48      1667160.94      6975540.26
      1666457.58      6976632.28      1664788.32      6976854.64
      1664105.07      6978208.03      1664558.55      6979636.53
      1666599.95      6981490.55      1663720.22      6981737.48
      1662032.15      6980887.71      1659868.40      6981624.70
      1660603.92      6984077.45      1659118.36      6984974.65
      1657464.11      6987781.27      1658199.49      6989432.73
      1654108.54      6989289.46      1654502.94      6992832.14
      1653849.89      6994432.89      1652598.83      6994695.86
      1652254.64      6995458.15      1653799.82      6996393.44
      1654254.88      6997572.95      1652905.00      6997988.00

Type RM Length L Ch R = 1,67896,410,410,410
BEGIN DESCRIPTION:
Swager Creek 117.0
END DESCRIPTION:
XS GIS Cut Line= 3
      1681366.77      6971555.88      1682253.95      6971598.42
      1683290.20      6971684.33
#Sta/Elev= 30
  4111.8 1814.49  4140.1 1814.10  4200.1 1811.36  4320.3 1807.69  4518.1 1803.07
  4617.1 1800.38  4730.7 1797.75  4740.7 1797.32  4750.8 1795.79  4770.8 1797.66
  4800.8 1797.58  4820.8 1796.26  4916.7 1797.42  4971.0 1796.53  4991.0 1795.06
  4998.0 1793.50  5009.0 1792.74  5009.3 1792.24  5013.2 1792.74  5021.1 1792.81
  5050.8 1798.91  5060.7 1799.82  5112.3 1801.56  5151.6 1803.79  5181.7 1804.54
  5349.7 1806.16  5458.0 1807.32  5626.9 1808.66  5700.0 1809.75  6039.8 1816.37
#Mann=12,-1,0
  4111.8   0.035       0  4518.1    0.16       0  4617.1    0.07       0
  4916.7   0.035       0  5009.0   0.035       0  5013.2   0.035       0
  5060.7    0.07       0  5112.3   0.035       0  5349.7    0.07       0
  5458.0   0.035       0  5626.9    0.07       0  5700.0   0.035       0
Bank Sta=5009,5013.2
Exp/Cntr=0.3,0.1

Type RM Length L Ch R = 1,67486,819,819,819
BEGIN DESCRIPTION:
Mapping XS cf5b50e2
END DESCRIPTION:
XS GIS Cut Line= 3
      1681088.34      6971816.64      1682255.01      6972007.62
      1683000.79      6972420.40
#Sta/Elev= 30
  3817.8 1819.52  3834.7 1817.91  3925.9 1813.85  4189.3 1805.64  4280.7 1803.57
  4401.4 1800.83  4645.3 1795.55  4701.1 1795.01  4736.5 1794.44  4766.9 1792.74
  4817.6 1794.65  4959.5 1795.15  4973.0 1794.59  4995.4 1791.59  4995.7 1791.09
  4999.3 1791.09  4999.6 1791.59  5008.4 1792.29  5014.1 1791.95  5022.8 1793.97
  5030.2 1797.12  5035.9 1797.14  5045.7 1799.10  5112.4 1801.79  5295.8 1806.41
  5507.7 1810.34  5617.2 1813.06  5640.0 1814.28  5765.8 1817.08  5852.4 1820.09
#Mann=7,-1,0
  3817.8   0.035       0  4280.7    0.07       0  4401.4   0.035       0
  4701.1    0.07       0  4995.4    0.07       0  4999.6    0.07       0
  5112.4   0.035       0
Bank Sta=4995.4,4999.6
Exp/Cntr=0.3,0.1

Type RM Length L Ch R = 1,66667,1234,1234,1234
BEGIN DESCRIPTION:
Mapping XS 35b3bb63
END DESCRIPTION:
XS GIS Cut Line= 3
      1680821.71      6972128.82      1681849.45      6972649.63
      1682627.24      6972687.82
#Sta/Elev= 30
  3841.9 1820.87  3867.8 1820.08  3968.9 1813.66  4036.2 1810.70  4068.3 1810.43
  4125.9 1808.14  4313.3 1803.78  4439.8 1800.16  4446.9 1799.18  4497.1 1798.44
  4596.7 1794.50  4754.1 1790.80  4807.1 1790.14  4876.2 1789.79  4936.9 1789.74
  4953.6 1788.15  4975.8 1787.91  4979.3 1786.80  4979.6 1786.30  4983.6 1786.80
  4985.7 1786.87  4994.1 1786.98  4999.6 1788.63  5085.5 1789.40  5227.0 1793.23
  5310.0 1795.11  5349.5 1796.71  5430.1 1801.47  5467.9 1802.81  5772.8 1809.85
#Mann=10,-1,0
  3841.9   0.035       0  4754.1    0.16       0  4807.1    0.07       0
  4876.2   0.035       0  4979.3    0.07       0  4983.6   0.035       0
  4985.7    0.07       0  5085.5   0.035       0  5227.0    0.07       0
  5349.5   0.035       0
Bank Sta=4979.3,4983.6
Exp/Cntr=0.3,0.1

Type RM Length L Ch R = 1,65433,947,947,947
BEGIN DESCRIPTION:
Mapping XS 3ded24b0
END DESCRIPTION:
XS GIS Cut Line= 3
      1680737.67      6972351.40      1681570.98      6973514.56
      1682105.43      6973903.25
#Sta/Elev= 30
  3564.1 1813.56  3573.2 1811.61  3617.4 1808.98  3739.0 1803.34  3822.8 1800.67
  3894.4 1798.64  4011.7 1795.12  4103.9 1794.54  4234.1 1789.86  4492.0 1786.33
  4605.5 1782.99  4835.9 1784.72  4957.5 1783.39  4993.2 1781.07  5011.7 1780.98
  5012.0 1780.48  5016.1 1780.98  5028.6 1783.39  5057.9 1781.75  5179.3 1783.92
  5208.6 1783.51  5222.5 1782.31  5244.2 1783.00  5250.4 1784.48  5272.0 1786.42
  5365.5 1790.58  5401.1 1795.99  5436.6 1798.18  5486.8 1799.98  5655.8 1803.06
#Mann=5,-1,0
  3564.1   0.035       0  3822.8    0.07       0  3894.4   0.035       0
  5011.7   0.035       0  5016.1   0.035       0
Bank Sta=5011.7,5016.1
Exp/Cntr=0.3,0.1

Type RM Length L Ch R = 1,64486,705,705,705
BEGIN DESCRIPTION:
Mapping XS cc5e915e
END DESCRIPTION:
XS GIS Cut Line= 3
      1680621.79      6972458.10      1680962.07      6973798.36
      1681083.59      6974638.64
#Sta/Elev= 30
  3627.4 1808.03  3632.5 1807.86  3703.0 1804.59  3738.8 1802.08  3813.0 1799.11
  4009.0 1793.24  4040.0 1791.54  4132.8 1783.69  4260.3 1781.55  4414.0 1778.55
  4470.8 1777.74  4509.8 1778.14  4625.7 1779.08  4721.7 1779.63  4803.6 1778.92
  4813.8 1777.65  4834.2 1777.06  4875.2 1777.09  4921.3 1778.38  4986.5 1776.64
  4986.9 1776.14  4991.8 1776.64  5060.3 1779.24  5110.9 1780.19  5201.0 1784.04
  5333.1 1787.53  5434.2 1794.53  5487.3 1796.12  5747.4 1800.20  5859.2 1803.13
#Mann=8,-1,0
  3627.4    0.07       0  3632.5   0.035       0  4260.3    0.07       0
  4414.0   0.035       0  4509.8    0.07       0  4625.7   0.035       0
  4986.5   0.035       0  4991.8   0.035       0
Bank Sta=4986.5,4991.8
Exp/Cntr=0.3,0.1

Type RM Length L Ch R = 1,63781,1332,1332,1332
BEGIN DESCRIPTION:
Mapping XS 7347ef94
END DESCRIPTION:
XS GIS Cut Line= 3
      1680465.54      6972367.80      1680347.48      6973551.83
      1680420.38      6974513.37
#Sta/Elev= 30
  3821.8 1810.42  3892.4 1807.58  3962.7 1803.87  3978.1 1802.33  4032.9 1800.02
  4167.7 1794.70  4244.1 1790.54  4324.5 1781.97  4364.7 1778.33  4387.9 1777.49
  4455.1 1774.54  4555.6 1773.53  4656.1 1773.65  4736.5 1775.29  4877.2 1776.30
  4888.9 1775.40  4937.5 1775.44  5015.2 1773.40  5015.6 1772.90  5020.5 1773.40
  5037.9 1774.16  5078.1 1777.76  5509.3 1786.97  5719.9 1793.14  5729.9 1794.45
  5760.0 1792.82  5780.1 1792.86  5800.1 1794.55  5890.4 1795.96  5976.0 1798.49
#Mann=6,-1,0
  3821.8    0.07       0  4032.9   0.035       0  4167.7    0.07       0
  4387.9   0.035       0  5015.2   0.035       0  5020.5   0.035       0
Bank Sta=5015.2,5020.5
Exp/Cntr=0.3,0.1

Type RM Length L Ch R = 1,62449,835,835,835
BEGIN DESCRIPTION:
Mapping XS cc383341
END DESCRIPTION:
XS GIS Cut Line= 3
      1680361.35      6972336.57      1679854.43      6972850.44
      1679364.85      6974492.79
#Sta/Elev= 30
  4297.1 1807.66  4570.0 1795.90  4597.4 1794.93  4769.3 1789.42  4811.7 1786.15
  4840.0 1782.44  4861.2 1780.83  4896.6 1775.99  4946.0 1771.86  4953.2 1769.69
  4985.7 1767.39  4986.2 1766.89  4991.2 1767.39  4998.6 1768.53  5033.2 1771.22
  5110.3 1770.65  5209.4 1771.54  5287.7 1770.13  5352.5 1770.11  5418.8 1771.96
  5633.4 1772.75  5673.8 1774.62  5738.1 1775.45  5909.1 1779.68  6046.9 1785.31
  6366.2 1792.83  6552.6 1798.48  6578.1 1799.41  6686.0 1803.80  6732.7 1807.42
#Mann=8,-1,0
  4297.1    0.07       0  4570.0   0.035       0  4597.4    0.07       0
  4985.7   0.035       0  4991.2    0.07       0  4998.6   0.035       0
  6552.6    0.07       0  6578.1   0.035       0
Bank Sta=4985.7,4991.2
Exp/Cntr=0.3,0.1

Type RM Length L Ch R = 1,61614,927,927,927
BEGIN DESCRIPTION:
Mapping XS d346481d
END DESCRIPTION:
XS GIS Cut Line= 3
      1679299.51      6972026.76      1679362.01      6973143.96
      1679302.11      6974209.03
#Sta/Elev= 30
  3887.0 1795.72  3894.5 1794.96  3991.1 1790.65  4054.5 1788.53  4098.6 1787.27
  4253.9 1779.54  4499.2 1773.05  4659.4 1770.20  4879.8 1768.34  4967.5 1765.67
  4979.9 1765.98  4990.0 1765.42  5038.4 1766.69  5060.1 1766.50  5097.2 1765.11
  5097.7 1764.61  5102.6 1764.61  5103.0 1765.11  5160.2 1768.25  5340.5 1774.30
  5440.7 1777.08  5450.7 1778.04  5460.7 1777.78  5641.0 1784.81  5662.2 1784.97
  5702.0 1786.23  5871.4 1790.11  5921.4 1791.89  6011.6 1793.79  6072.7 1795.96
#Mann=7,-1,0
  3887.0   0.035       0  3991.1    0.07       0  4054.5   0.035       0
  5097.2   0.035       0  5103.0   0.035       0  5662.2    0.07       0
  5702.0   0.035       0
Bank Sta=5097.2,5103
Exp/Cntr=0.3,0.1

Type RM Length L Ch R = 1,60687,962,962,962
BEGIN DESCRIPTION:
Mapping XS d8a52e3a
END DESCRIPTION:
XS GIS Cut Line= 3
      1679051.05      6971801.47      1678564.96      6973058.37
      1678693.30      6974494.42
#Sta/Elev= 30
  3660.4 1800.07  3668.0 1799.36  3741.8 1798.73  3861.6 1794.64  3935.3 1793.80
  3978.3 1791.58  4049.7 1789.86  4149.9 1785.83  4297.8 1781.85  4327.7 1780.56
  4417.9 1773.27  4466.7 1770.63  4739.4 1765.17  4829.2 1762.61  4883.7 1762.31
  4938.3 1763.17  4962.9 1762.42  4983.2 1760.64  4983.7 1760.14  4989.1 1760.64
  5063.8 1763.61  5395.6 1770.46  5527.1 1773.39  5611.7 1775.11  5651.2 1776.15
  6061.8 1785.43  6217.6 1790.08  6278.6 1791.84  6382.5 1795.62  6449.8 1798.40
#Mann=10,-1,0
  3660.4   0.035       0  4983.2   0.035       0  4989.1   0.035       0
  5395.6    0.07       0  5527.1   0.035       0  5611.7    0.07       0
  5651.2   0.035       0  6217.6    0.07       0  6278.6   0.035       0
  6382.5    0.07       0
Bank Sta=4983.2,4989.1
Exp/Cntr=0.3,0.1

Type RM Length L Ch R = 1,59725,865,865,865
BEGIN DESCRIPTION:
Mapping XS feb578b1
END DESCRIPTION:
XS GIS Cut Line= 3
      1677742.05      6971468.10      1678054.54      6972544.48
      1677926.07      6974377.86
#Sta/Elev= 30
  3881.5 1802.36  4006.3 1793.97  4180.8 1786.02  4402.0 1779.24  4610.3 1775.12
  4732.5 1768.14  4737.7 1766.63  4949.4 1762.38  4983.0 1758.06  5015.9 1756.01
  5035.9 1758.28  5064.1 1759.18  5176.3 1755.93  5196.3 1757.46  5213.3 1755.47
  5213.8 1754.97  5219.5 1755.47  5256.5 1759.37  5286.5 1760.44  5346.7 1758.62
  5416.9 1760.91  5611.0 1763.11  5904.8 1767.40  6002.7 1766.60  6100.6 1770.81
  6376.1 1778.42  6579.7 1784.61  6641.0 1787.85  6786.1 1795.34  6840.2 1798.20
#Mann=11,-1,0
  3881.5    0.07       0  4180.8   0.035       0  5213.3   0.035       0
  5219.5   0.035       0  5611.0    0.16       0  5904.8   0.035       0
  6002.7    0.07       0  6100.6   0.035       0  6376.1    0.07       0
  6641.0   0.035       0  6786.1    0.07       0
Bank Sta=5213.3,5219.5
Exp/Cntr=0.3,0.1

Type RM Length L Ch R = 1,58860,530,530,530
BEGIN DESCRIPTION:
Mapping XS d8d965c1
END DESCRIPTION:
XS GIS Cut Line= 3
      1677367.04      6971492.41      1677436.49      6973009.76
      1677495.51      6974172.92
#Sta/Elev= 30
  3484.2 1807.60  3529.8 1803.88  3609.9 1794.00  3650.0 1791.51  3670.0 1789.04
  3766.4 1783.96  4099.1 1772.16  4580.9 1756.97  4691.1 1756.47  4761.1 1753.08
  4831.2 1756.33  4901.3 1756.34  4961.3 1754.86  4981.4 1752.24  4996.6 1751.89
  4997.1 1751.39  5002.9 1751.89  5041.4 1755.18  5121.5 1755.19  5191.6 1758.32
  5251.7 1757.65  5311.8 1759.71  5331.8 1761.95  5391.9 1762.89  5559.1 1769.04
  5601.9 1770.56  5832.4 1779.13  5932.6 1784.15  6072.8 1796.76  6167.8 1801.40
#Mann=6,-1,0
  3484.2    0.07       0  4099.1   0.035       0  4996.6   0.035       0
  5002.9   0.035       0  5559.1    0.07       0  5601.9   0.035       0
Bank Sta=4996.6,5002.9
Exp/Cntr=0.3,0.1

Type RM Length L Ch R = 1,58330,860,860,860
BEGIN DESCRIPTION:
Mapping XS 91609e7f
END DESCRIPTION:
XS GIS Cut Line= 3
      1676655.24      6971619.15      1677033.71      6973296.22
      1677252.46      6974139.98
#Sta/Elev= 30
  3289.1 1787.61  3369.9 1782.97  3580.6 1774.95  3614.3 1773.64  3667.2 1772.45
  3716.5 1769.82  3728.7 1770.40  3790.2 1769.09  3830.8 1767.08  3851.2 1765.92
  3892.8 1766.31  4260.7 1757.08  4443.8 1754.87  4876.9 1753.58  4917.9 1752.93
  4958.9 1750.47  4977.0 1750.85  5017.2 1749.97  5017.7 1749.47  5023.9 1749.97
  5034.7 1750.38  5041.2 1752.03  5123.8 1757.03  5185.8 1758.77  5264.0 1764.69
  5599.2 1778.67  5702.3 1783.25  5743.7 1786.99  5870.4 1795.54  5880.0 1795.74
#Mann=10,-1,0
  3289.1    0.07       0  3580.6   0.035       0  3614.3    0.07       0
  3830.8   0.035       0  4977.0    0.07       0  5017.2    0.07       0
  5023.9    0.07       0  5264.0   0.035       0  5599.2    0.07       0
  5870.4   0.035       0
Bank Sta=5017.2,5023.9
Exp/Cntr=0.3,0.1

Type RM Length L Ch R = 1,57470,926,926,926
BEGIN DESCRIPTION:
Mapping XS 5e116441
END DESCRIPTION:
XS GIS Cut Line= 3
      1675617.05      6972025.39      1676276.76      6973188.58
      1677037.15      6974070.48
#Sta/Elev= 30
  3663.4 1796.28  3723.9 1789.10  3773.2 1779.88  3824.8 1774.67  3982.1 1764.85
  4104.5 1760.02  4139.6 1759.19  4193.8 1755.16  4252.1 1751.98  4336.7 1751.96
  4465.2 1746.97  4534.3 1745.75  4534.8 1745.25  4541.1 1745.75  4625.4 1746.31
  4684.7 1747.02  4768.0 1747.59  4925.7 1749.01  4969.0 1746.30  5006.4 1745.98
  5020.1 1746.64  5098.2 1750.64  5112.5 1753.80  5204.6 1757.29  5374.7 1760.84
  5403.2 1764.13  5460.2 1766.69  5765.2 1772.47  5972.1 1778.10  6165.1 1783.34
#Mann=15,-1,0
  3663.4    0.07       0  3824.8   0.035       0  3982.1    0.07       0
  4104.5   0.035       0  4193.8    0.07       0  4336.7   0.035       0
  4465.2    0.07       0  4534.3   0.035       0  4541.1    0.07       0
  4625.4   0.035       0  4684.7    0.07       0  4768.0   0.035       0
  5006.4    0.07       0  5020.1   0.035       0  5972.1    0.07       0
Bank Sta=4534.3,4541.1
Exp/Cntr=0.3,0.1

Type RM Length L Ch R = 1,56544,625,625,625
BEGIN DESCRIPTION:
Mapping XS af363246
END DESCRIPTION:
XS GIS Cut Line= 3
      1674884.86      6972478.19      1675515.05      6973131.81
      1676496.40      6973863.26
#Sta/Elev= 30
  4094.8 1792.89  4158.4 1788.79  4172.6 1788.17  4179.5 1789.18  4229.2 1783.36
  4236.1 1783.65  4243.3 1781.85  4250.3 1782.11  4257.5 1780.06  4278.6 1778.57
  4285.8 1776.44  4292.7 1776.64  4328.2 1771.80  4538.6 1756.44  4575.7 1752.30
  4618.2 1750.10  4830.9 1742.13  4865.6 1740.33  5003.0 1738.40  5003.3 1738.19
  5003.8 1737.69  5010.4 1738.19  5065.0 1738.38  5121.5 1742.29  5257.0 1746.92
  5763.7 1756.44  5963.9 1762.15  6013.9 1765.28  6107.8 1768.35  6226.7 1769.23
#Mann=6,-1,0
  4094.8    0.07       0  4538.6   0.035       0  4830.9    0.07       0
  5003.0   0.035       0  5003.3    0.07       0  5010.4   0.035       0
Bank Sta=5003.3,5010.4
Exp/Cntr=0.3,0.1

Type RM Length L Ch R = 1,55919,701,701,701
BEGIN DESCRIPTION:
Mapping XS 408d7648
END DESCRIPTION:
XS GIS Cut Line= 3
      1674452.53      6972603.14      1674952.55      6973301.08
      1675732.99      6974604.42
#Sta/Elev= 30
  4147.9 1783.86  4160.4 1782.89  4231.6 1770.91  4282.0 1765.03  4474.8 1755.10
  4589.2 1751.01  4711.9 1744.69  4741.0 1744.17  4838.9 1739.27  4848.2 1738.25
  4877.7 1738.39  4904.7 1735.96  4934.2 1733.20  4961.6 1732.43  4995.7 1730.88
  4996.2 1730.38  5002.9 1730.88  5020.7 1732.16  5094.6 1732.16  5137.3 1736.45
  5196.0 1738.90  5311.9 1740.56  5508.7 1742.12  5625.4 1741.95  5748.8 1740.24
  5932.6 1745.99  6145.7 1750.76  6390.6 1757.76  6411.5 1758.46  6525.6 1762.20
#Mann=14,-1,0
  4147.9    0.07       0  4589.2   0.035       0  4741.0    0.07       0
  4838.9   0.035       0  4904.7    0.07       0  4961.6   0.035       0
  4995.7   0.035       0  5002.9   0.035       0  5196.0    0.07       0
  5311.9   0.035       0  5932.6    0.07       0  6145.7   0.035       0
  6390.6    0.07       0  6411.5   0.035       0
Bank Sta=4995.7,5002.9
Exp/Cntr=0.3,0.1

Type RM Length L Ch R = 1,55218,637,637,637
BEGIN DESCRIPTION:
Mapping XS edc5f9fe
END DESCRIPTION:
XS GIS Cut Line= 3
      1673845.76      6973058.00      1674361.40      6973589.27
      1675375.73      6974754.46
#Sta/Elev= 30
  4258.9 1776.47  4293.7 1773.68  4307.9 1770.02  4329.0 1768.63  4336.2 1766.98
  4392.7 1763.45  4676.0 1753.64  4712.8 1752.24  4753.4 1748.36  4795.8 1742.21
  4905.0 1736.37  4933.1 1734.18  4993.9 1729.17  4998.3 1727.34  5018.7 1723.29
  5019.2 1722.79  5026.4 1723.29  5084.2 1727.79  5114.6 1727.96  5164.0 1731.88
  5199.1 1733.06  5516.7 1737.38  5615.1 1738.60  5966.2 1743.43  5998.6 1743.93
  6118.8 1746.44  6262.5 1750.58  6348.0 1755.62  6489.2 1758.56  6544.1 1759.57
#Mann=14,-1,0
  4258.9    0.07       0  4676.0   0.035       0  4712.8    0.07       0
  4905.0   0.035       0  4933.1    0.07       0  5018.7    0.07       0
  5026.4    0.07       0  5084.2   0.035       0  5516.7    0.16       0
  5615.1    0.07       0  5966.2   0.035       0  5998.6    0.07       0
  6118.8   0.035       0  6489.2    0.07       0
Bank Sta=5018.7,5026.4
Exp/Cntr=0.3,0.1

Type RM Length L Ch R = 1,54581,636,636,636
BEGIN DESCRIPTION:
Mapping XS 3e509a5e
END DESCRIPTION:
XS GIS Cut Line= 3
      1673593.81      6973277.60      1673898.51      6973988.58
      1674382.32      6975364.58
#Sta/Elev= 30
  4231.5 1760.89  4294.9 1755.36  4343.5 1752.81  4429.1 1749.53  4499.8 1744.21
  4546.9 1742.06  4719.6 1737.03  4886.0 1730.36  4927.7 1725.75  4939.1 1723.36
  4976.4 1720.77  4976.9 1720.27  4984.3 1720.77  4993.5 1721.76  5002.0 1724.52
  5007.3 1724.52  5009.6 1725.91  5015.0 1726.60  5032.6 1726.37  5066.3 1726.05
  5184.6 1729.40  5345.0 1730.94  5520.3 1728.91  5551.2 1730.33  5629.8 1731.02
  5683.7 1733.68  5714.6 1735.50  6096.5 1747.27  6434.8 1758.66  6463.6 1759.45
#Mann=9,-1,0
  4231.5    0.07       0  4343.5   0.035       0  4719.6    0.07       0
  4976.4    0.07       0  4984.3    0.07       0  5032.6   0.035       0
  5683.7    0.07       0  6096.5   0.035       0  6434.8    0.07       0
Bank Sta=4976.4,4984.3
Exp/Cntr=0.3,0.1

Type RM Length L Ch R = 1,53945,654,654,654
BEGIN DESCRIPTION:
Mapping XS daa1b1e6
END DESCRIPTION:
XS GIS Cut Line= 3
      1673267.87      6973346.89      1673361.62      6974247.91
      1673447.55      6975328.62
#Sta/Elev= 30
  4104.4 1757.11  4135.7 1753.50  4175.9 1750.26  4226.4 1747.44  4314.9 1740.55
  4320.0 1740.78  4413.5 1735.17  4497.6 1731.25  4670.7 1725.78  4802.8 1723.45
  4929.9 1723.03  4995.0 1719.67  5003.9 1717.46  5004.4 1716.96  5011.8 1717.46
  5020.4 1717.52  5040.5 1722.30  5050.5 1722.76  5120.9 1723.03  5170.9 1720.99
  5201.0 1724.26  5271.2 1728.48  5403.1 1732.53  5467.4 1734.17  5538.6 1736.40
  5652.0 1740.06  5752.7 1744.30  5942.9 1750.90  6013.5 1753.56  6094.4 1758.41
#Mann=9,-1,0
  4104.4    0.07       0  4670.7   0.035       0  5003.9   0.035       0
  5011.8   0.035       0  5403.1    0.07       0  5467.4   0.035       0
  5538.6    0.07       0  5652.0   0.035       0  5942.9    0.07       0
Bank Sta=5003.9,5011.8
Exp/Cntr=0.3,0.1

Type RM Length L Ch R = 1,53291,747,747,747
BEGIN DESCRIPTION:
Mapping XS cec0900c
END DESCRIPTION:
XS GIS Cut Line= 3
      1672872.54      6973393.32      1672785.73      6974241.87
      1672844.20      6974984.60
#Sta/Elev= 30
  4151.0 1748.67  4206.0 1744.88  4266.3 1739.68  4296.4 1735.87  4372.2 1729.17
  4468.5 1724.80  4497.5 1723.41  4572.6 1721.89  4668.8 1720.74  4738.7 1720.33
  4819.1 1717.60  4900.8 1718.83  4958.5 1718.60  4969.9 1716.18  4990.0 1714.10
  5006.0 1713.58  5006.5 1713.08  5013.8 1713.08  5014.3 1713.58  5020.2 1713.70
  5056.8 1721.56  5061.8 1720.46  5080.3 1723.62  5128.8 1725.80  5314.6 1730.29
  5361.2 1732.30  5391.3 1732.44  5501.6 1736.21  5561.8 1739.73  5749.0 1743.17
#Mann=8,-1,0
  4151.0    0.07       0  4468.5   0.035       0  4572.6    0.07       0
  4668.8   0.035       0  4900.8    0.07       0  5006.0    0.07       0
  5014.3    0.07       0  5128.8   0.035       0
Bank Sta=5006,5014.3
Exp/Cntr=0.3,0.1

Type RM Length L Ch R = 1,52544,758,758,758
BEGIN DESCRIPTION:
Mapping XS f6fc4760
END DESCRIPTION:
XS GIS Cut Line= 3
      1671799.18      6972999.72      1672111.69      6974048.38
      1672566.56      6975208.13
#Sta/Elev= 30
  3916.3 1749.55  3957.8 1746.27  4050.2 1742.34  4123.2 1736.87  4134.1 1735.03
  4206.7 1730.38  4369.3 1723.83  4408.3 1722.41  4518.4 1717.34  4571.9 1716.18
  4603.2 1716.81  4619.2 1715.56  4652.3 1714.77  4718.0 1716.18  4890.3 1715.07
  4971.6 1714.18  4995.3 1710.89  4995.8 1710.39  5003.8 1710.89  5033.8 1712.15
  5089.4 1712.14  5096.1 1712.51  5113.8 1715.52  5246.3 1721.23  5506.6 1724.41
  5691.4 1727.42  5848.0 1731.03  5990.0 1736.88  6106.3 1739.40  6256.3 1741.30
#Mann=11,-1,0
  3916.3    0.07       0  4369.3   0.035       0  4408.3    0.07       0
  4518.4   0.035       0  4890.3    0.07       0  4995.3    0.07       0
  5003.8    0.07       0  5033.8   0.035       0  5246.3    0.16       0
  5506.6   0.035       0  5990.0    0.07       0
Bank Sta=4995.3,5003.8
Exp/Cntr=0.3,0.1

Type RM Length L Ch R = 1,51786,877,877,877
BEGIN DESCRIPTION:
Mapping XS d50c1b23
END DESCRIPTION:
XS GIS Cut Line= 3
      1671389.47      6973256.67      1671382.52      6973944.21
      1671444.96      6975664.70
#Sta/Elev= 30
  4318.6 1754.41  4369.9 1753.07  4419.9 1750.04  4499.9 1742.32  4659.9 1733.55
  4719.9 1728.01  4929.3 1713.81  4960.0 1707.63  4990.0 1708.39  5001.1 1706.04
  5001.6 1705.54  5010.0 1706.04  5050.0 1708.58  5112.4 1708.85  5160.1 1706.36
  5248.3 1709.12  5290.1 1710.90  5420.2 1712.07  5540.3 1708.91  5621.2 1712.11
  5650.4 1712.83  5670.4 1714.81  5770.5 1714.67  5843.9 1717.75  6110.7 1725.02
  6209.1 1729.20  6300.8 1731.73  6472.4 1733.50  6571.1 1734.57  6727.8 1738.11
#Mann=11,-1,0
  4318.6    0.07       0  4929.3   0.035       0  5001.1   0.035       0
  5010.0   0.035       0  5112.4    0.07       0  5248.3   0.035       0
  5621.2    0.07       0  5843.9   0.035       0  6209.1    0.07       0
  6472.4   0.035       0  6571.1    0.07       0
Bank Sta=5001.1,5010
Exp/Cntr=0.3,0.1

Type RM Length L Ch R = 1,50909,812,812,812
BEGIN DESCRIPTION:
Mapping XS 64ccbb03
END DESCRIPTION:
XS GIS Cut Line= 3
      1670212.36      6973581.68      1670646.41      6974102.54
      1671222.81      6975192.84
#Sta/Elev= 30
  4326.2 1728.59  4382.5 1722.89  4438.6 1715.39  4489.2 1711.89  4524.4 1708.09
  4586.1 1706.27  4737.9 1704.54  4801.6 1701.91  4857.6 1703.12  4914.9 1702.82
  4921.4 1703.62  4929.2 1702.67  4972.2 1701.22  5025.9 1700.69  5026.4 1700.19
  5034.8 1700.69  5066.9 1701.37  5102.0 1700.86  5118.4 1701.96  5250.4 1704.54
  5288.8 1706.48  5294.4 1705.65  5332.8 1708.30  5354.8 1707.91  5454.5 1710.13
  5525.2 1712.34  5657.9 1713.90  5761.7 1715.42  5954.1 1719.89  6237.5 1730.06
#Mann=6,-1,0
  4326.2    0.07       0  4586.1   0.035       0  5025.9   0.035       0
  5034.8   0.035       0  5454.5    0.07       0  5657.9   0.035       0
Bank Sta=5025.9,5034.8
Exp/Cntr=0.3,0.1

Type RM Length L Ch R = 1,50097,575,575,575
BEGIN DESCRIPTION:
Mapping XS 2dc74303
END DESCRIPTION:
XS GIS Cut Line= 3
      1669677.65      6973987.95      1669948.49      6974390.74
      1670528.37      6975619.94
#Sta/Elev= 30
  4511.6 1710.04  4531.7 1709.73  4639.7 1704.59  4776.8 1699.70  4834.7 1697.92
  4933.7 1697.02  4942.7 1695.60  4948.7 1693.24  4973.9 1692.24  4974.4 1691.74
  4983.5 1692.24  4984.7 1693.22  4992.3 1693.68  5041.9 1695.73  5073.0 1695.93
  5119.4 1697.26  5142.2 1697.17  5222.6 1695.14  5256.1 1696.30  5278.8 1698.34
  5339.7 1700.31  5347.5 1700.66  5428.8 1702.62  5647.5 1707.39  5887.7 1712.25
  5938.7 1714.15  5955.9 1715.53  5961.4 1716.71  6029.8 1720.03  6356.1 1726.05
#Mann=11,-1,0
  4511.6   0.035       0  4973.9   0.035       0  4983.5   0.035       0
  5041.9    0.07       0  5073.0   0.035       0  5222.6    0.07       0
  5339.7   0.035       0  5347.5    0.07       0  5428.8   0.035       0
  5647.5    0.07       0  5887.7   0.035       0
Bank Sta=4973.9,4983.5
Exp/Cntr=0.3,0.1

Type RM Length L Ch R = 1,49522,663,663,663
BEGIN DESCRIPTION:
Swager Creek 82.0
END DESCRIPTION:
XS GIS Cut Line= 3
      1669566.55      6974052.22      1669655.00      6974838.00
      1669896.40      6975751.81
#Sta/Elev= 30
  4214.1 1707.85  4254.8 1706.84  4350.5 1703.95  4599.9 1694.77  4781.9 1693.85
  4864.0 1691.34  4884.1 1693.61  4904.2 1693.39  4945.0 1691.34  4969.7 1687.17
  4970.2 1686.67  4979.6 1687.17  4994.8 1687.29  5034.8 1691.82  5046.2 1692.80
  5062.7 1691.56  5087.6 1691.43  5138.0 1693.40  5295.8 1697.71  5304.8 1697.36
  5346.2 1699.39  5379.6 1699.28  5449.6 1703.23  5501.3 1711.65  5535.5 1714.32
  5631.5 1716.43  5736.7 1718.97  5807.0 1721.98  5884.9 1723.62  5950.0 1724.86
#Mann=13,-1,0
  4214.1   0.035       0  4254.8    0.07       0  4350.5   0.035       0
  4781.9    0.07       0  4945.0   0.035       0  4969.7   0.035       0
  4979.6   0.035       0  5034.8    0.07       0  5138.0   0.035       0
  5295.8    0.07       0  5631.5   0.035       0  5736.7    0.07       0
  5884.9   0.035       0
Bank Sta=4969.7,4979.6
Exp/Cntr=0.3,0.1

Type RM Length L Ch R = 1,48859,702,702,702
BEGIN DESCRIPTION:
Mapping XS fd823527
END DESCRIPTION:
XS GIS Cut Line= 3
      1669472.80      6974128.56      1669292.24      6975343.86
      1669434.61      6976302.21
#Sta/Elev= 30
  3778.7 1705.56  4003.8 1701.38  4142.6 1695.54  4495.0 1691.94  4705.5 1689.95
  4955.2 1688.41  4981.6 1685.90  5001.4 1683.37  5016.6 1683.36  5017.1 1682.86
  5026.7 1683.36  5072.2 1690.49  5102.5 1693.53  5122.7 1697.09  5128.0 1699.11
  5142.9 1701.23  5197.4 1707.12  5203.6 1709.06  5261.7 1711.37  5274.4 1712.74
  5294.6 1712.94  5400.6 1712.88  5457.7 1711.49  5470.0 1712.02  5534.3 1709.92
  5597.9 1711.33  5648.4 1715.21  5850.6 1725.28  5949.7 1733.67  5976.2 1736.30
#Mann=8,-1,0
  3778.7   0.035       0  4495.0    0.07       0  4705.5   0.035       0
  4981.6    0.07       0  5016.6    0.07       0  5026.7    0.07       0
  5457.7   0.035       0  5949.7    0.07       0
Bank Sta=5016.6,5026.7
Exp/Cntr=0.3,0.1

Type RM Length L Ch R = 1,48157,847,847,847
BEGIN DESCRIPTION:
Swager Creek 81.0
END DESCRIPTION:
XS GIS Cut Line= 3
      1669420.73      6974132.03      1668705.00      6975438.00
      1668868.69      6976327.73
#Sta/Elev= 30
  3511.0 1705.42  3865.9 1697.84  4019.8 1695.96  4239.7 1693.84  4279.3 1692.06
  4338.8 1692.73  4510.6 1689.49  4678.5 1687.24  4829.2 1684.78  4942.9 1684.75
  4986.5 1683.19  5010.4 1680.98  5015.4 1679.43  5015.9 1678.93  5025.7 1679.43
  5026.8 1680.64  5031.8 1679.58  5079.8 1690.53  5084.9 1689.94  5091.7 1692.07
  5112.1 1695.01  5138.0 1698.30  5143.0 1697.56  5182.5 1702.90  5244.1 1707.39
  5352.4 1710.34  5604.0 1719.69  5708.7 1723.58  5793.3 1726.22  5904.9 1733.14
#Mann=11,-1,0
  3511.0   0.035       0  4019.8    0.07       0  4239.7   0.035       0
  4510.6    0.07       0  4678.5   0.035       0  5015.4   0.035       0
  5025.7   0.035       0  5182.5    0.07       0  5352.4   0.035       0
  5604.0    0.07       0  5708.7   0.035       0
Bank Sta=5015.4,5025.7
Exp/Cntr=0.3,0.1

Type RM Length L Ch R = 1,47310,806,806,806
BEGIN DESCRIPTION:
Swager Creek 79.0
END DESCRIPTION:
XS GIS Cut Line= 3
      1667133.45      6974305.15      1668155.00      6975438.00
      1668760.53      6976348.63
#Sta/Elev= 30
  3479.7 1760.27  3560.9 1759.20  3581.8 1761.74  3596.0 1756.83  3638.6 1753.36
  3687.9 1742.41  3801.5 1729.39  3850.9 1718.61  3914.4 1709.73  4077.6 1696.19
  4279.0 1690.24  4679.7 1681.49  4920.3 1681.89  4955.4 1680.21  4969.6 1675.20
  5003.2 1674.34  5003.7 1673.84  5022.0 1674.34  5084.8 1687.45  5131.1 1690.67
  5233.7 1702.58  5247.9 1703.87  5356.2 1707.87  5419.6 1709.30  5475.8 1710.41
  5625.4 1714.41  5851.1 1718.01  6000.2 1722.22  6058.8 1723.92  6098.7 1728.23
#Mann=14,-1,0
  3479.7    0.07       0  4077.6   0.035       0  4279.0    0.07       0
  5003.2    0.07       0  5022.0    0.07       0  5131.1   0.035       0
  5233.7    0.07       0  5247.9   0.035       0  5356.2    0.07       0
  5419.6   0.035       0  5475.8    0.07       0  5625.4   0.035       0
  5851.1    0.07       0  6000.2   0.035       0
Bank Sta=5003.2,5022
Exp/Cntr=0.3,0.1

Type RM Length L Ch R = 1,46504,729,729,729
BEGIN DESCRIPTION:
Mapping XS 09a42c74
END DESCRIPTION:
XS GIS Cut Line= 3
      1666857.13      6974657.02      1667430.03      6975546.76
      1668167.88      6977230.78
#Sta/Elev= 30
  3952.2 1759.29  4004.1 1757.93  4088.5 1755.97  4155.1 1751.42  4218.5 1738.50
  4327.5 1723.75  4369.7 1715.98  4429.1 1709.56  4509.0 1697.12  4530.2 1692.14
  4759.2 1678.56  4805.5 1676.59  4901.0 1678.48  4941.5 1677.13  4971.9 1672.41
  4998.8 1671.97  4999.3 1671.47  5017.6 1671.97  5037.2 1672.17  5077.3 1678.71
  5636.4 1683.70  6032.3 1694.26  6159.0 1700.29  6334.2 1705.10  6375.2 1706.40
  6483.3 1711.39  6541.2 1714.81  6654.9 1727.32  6730.5 1732.11  6849.0 1746.05
#Mann=12,-1,0
  3952.2   0.035       0  4004.1    0.07       0  4759.2   0.035       0
  4901.0    0.07       0  4998.8    0.07       0  5017.6    0.07       0
  5077.3   0.035       0  6159.0    0.07       0  6334.2   0.035       0
  6375.2    0.07       0  6483.3   0.035       0  6541.2    0.07       0
Bank Sta=4998.8,5017.6
Exp/Cntr=0.3,0.1

Type RM Length L Ch R = 1,45775,576,576,576
BEGIN DESCRIPTION:
Mapping XS 1db3e654
END DESCRIPTION:
XS GIS Cut Line= 3
      1666527.25      6975043.27      1666809.37      6975794.15
      1667797.90      6977324.64
#Sta/Elev= 30
  4206.5 1743.94  4215.6 1745.82  4240.5 1744.52  4270.7 1745.78  4276.1 1747.62
  4457.2 1747.63  4489.3 1745.08  4536.5 1736.71  4587.4 1728.57  4637.2 1724.66
  4713.6 1714.30  4807.9 1704.77  4873.9 1692.14  4928.9 1684.89  5002.1 1679.10
  5029.6 1670.11  5056.5 1668.21  5057.0 1667.71  5075.4 1668.21  5085.8 1670.19
  5168.0 1674.07  5377.4 1671.75  5513.3 1677.52  5662.1 1680.09  6041.4 1686.76
  6204.5 1690.94  6349.2 1696.31  6577.5 1707.34  6722.7 1723.41  6830.6 1731.01
#Mann=9,-1,0
  4206.5    0.16       0  4536.5    0.07       0  5056.5    0.07       0
  5075.4    0.07       0  5085.8   0.035       0  5662.1    0.16       0
  6041.4    0.07       0  6204.5   0.035       0  6349.2    0.07       0
Bank Sta=5056.5,5075.4
Exp/Cntr=0.3,0.1

Type RM Length L Ch R = 1,45199,516,516,516
BEGIN DESCRIPTION:
Mapping XS 26cbbb34
END DESCRIPTION:
XS GIS Cut Line= 3
      1666266.76      6975401.81      1666600.09      6976290.68
      1667530.30      6977456.92
#Sta/Elev= 30
  4051.9 1708.03  4233.4 1707.75  4356.3 1703.90  4487.6 1698.62  4592.5 1691.38
  4715.8 1674.30  4744.1 1672.67  4768.3 1671.64  4873.9 1671.77  4941.8 1669.84
  4968.3 1666.70  4987.5 1665.69  4988.0 1665.19  5006.5 1665.69  5052.3 1668.31
  5101.9 1666.94  5166.0 1674.02  5230.7 1675.56  5289.0 1675.42  5366.1 1674.37
  5596.0 1679.97  5614.4 1680.71  5698.8 1682.17  5933.3 1687.73  5998.2 1689.71
  6037.9 1691.25  6213.0 1699.77  6290.1 1706.10  6354.1 1715.34  6493.0 1725.41
#Mann=18,-1,0
  4051.9    0.07       0  4356.3   0.035       0  4487.6    0.07       0
  4744.1   0.035       0  4768.3    0.07       0  4873.9   0.035       0
  4968.3    0.07       0  4987.5    0.07       0  5006.5    0.07       0
  5166.0   0.035       0  5230.7    0.07       0  5289.0    0.16       0
  5596.0   0.035       0  5614.4    0.16       0  5698.8   0.035       0
  5933.3    0.07       0  5998.2   0.035       0  6037.9    0.07       0
Bank Sta=4987.5,5006.5
Exp/Cntr=0.3,0.1

Type RM Length L Ch R = 1,44683,1049,1049,1049
BEGIN DESCRIPTION:
Mapping XS 6ed1704a
END DESCRIPTION:
XS GIS Cut Line= 3
      1664884.78      6975509.41      1666357.03      6976689.99
      1667310.93      6977678.57
#Sta/Elev= 30
  3121.2 1738.00  3191.4 1736.28  3313.1 1722.85  3418.7 1715.00  3532.3 1698.32
  3718.0 1685.33  3788.4 1670.10  3801.5 1669.13  4287.7 1673.65  4535.7 1668.74
  4841.6 1668.20  4913.4 1667.29  4967.9 1663.23  4968.4 1662.73  4987.0 1663.23
  4998.2 1667.75  5010.4 1667.61  5012.6 1669.69  5057.5 1670.94  5189.6 1672.97
  5315.7 1675.42  5360.3 1675.93  5476.9 1678.24  5729.6 1684.12  5856.6 1688.63
  5889.2 1690.32  6009.0 1695.18  6144.2 1703.58  6228.9 1713.25  6382.1 1723.23
#Mann=14,-1,0
  3121.2    0.07       0  3801.5   0.035       0  4841.6    0.07       0
  4967.9    0.07       0  4987.0    0.07       0  5057.5   0.035       0
  5189.6    0.07       0  5315.7   0.035       0  5360.3    0.16       0
  5476.9    0.07       0  5729.6   0.035       0  5856.6    0.07       0
  5889.2   0.035       0  6009.0    0.07       0
Bank Sta=4967.9,4987
Exp/Cntr=0.3,0.1

Type RM Length L Ch R = 1,43634,590,590,590
BEGIN DESCRIPTION:
Mapping XS dbf81c7c
END DESCRIPTION:
XS GIS Cut Line= 3
      1664696.62      6975721.94      1665453.56      6976548.32
      1666019.52      6978020.53
#Sta/Elev= 30
  3894.0 1741.27  4060.0 1735.11  4166.1 1723.47  4180.3 1724.64  4215.4 1720.56
  4343.1 1713.82  4364.0 1710.46  4399.8 1708.36  4406.6 1706.02  4477.5 1696.92
  4704.1 1676.94  4937.5 1670.00  4965.9 1666.40  4980.0 1662.43  4984.4 1658.28
  4984.9 1657.78  5004.0 1658.28  5105.7 1664.86  5398.0 1666.96  5625.0 1665.34
  5764.3 1666.64  6000.0 1673.20  6095.9 1679.14  6206.0 1687.84  6230.6 1693.48
  6260.6 1696.44  6285.3 1701.92  6484.6 1716.50  6509.2 1720.64  6591.9 1724.49
#Mann=7,-1,0
  3894.0    0.07       0  4704.1   0.035       0  4984.4   0.035       0
  5004.0   0.035       0  5105.7    0.07       0  5398.0   0.035       0
  6095.9    0.07       0
Bank Sta=4984.4,5004
Exp/Cntr=0.3,0.1

Type RM Length L Ch R = 1,43044,803,803,803
BEGIN DESCRIPTION:
Mapping XS df80b7a2
END DESCRIPTION:
XS GIS Cut Line= 3
      1664609.83      6976249.74      1664960.50      6976784.43
      1665515.78      6977943.57
#Sta/Elev= 30
  4364.2 1742.89  4541.2 1734.88  4568.2 1729.40  4589.3 1721.66  4619.5 1714.91
  4707.0 1702.42  4749.1 1693.08  4779.3 1690.12  4800.4 1685.67  4828.5 1683.76
  4864.4 1675.35  4914.9 1668.40  4930.0 1667.97  4962.3 1657.32  4962.8 1656.82
  4981.9 1657.32  4984.2 1658.06  5085.2 1663.42  5196.1 1661.42  5350.3 1663.21
  5572.3 1662.87  5630.7 1661.48  5761.2 1662.72  5866.4 1665.70  5908.2 1669.30
  5939.0 1675.76  5983.3 1680.03  6095.1 1698.52  6216.2 1710.10  6288.9 1719.35
#Mann=7,-1,0
  4364.2    0.07       0  4962.3   0.035       0  4981.9    0.07       0
  4984.2   0.035       0  5350.3    0.07       0  5572.3   0.035       0
  5866.4    0.07       0
Bank Sta=4962.3,4981.9
Exp/Cntr=0.3,0.1

Type RM Length L Ch R = 1,42241,750,750,750
BEGIN DESCRIPTION:
Mapping XS 817a2b56
END DESCRIPTION:
XS GIS Cut Line= 3
      1663992.12      6976985.14      1664707.38      6977370.54
      1665338.25      6977984.08
#Sta/Elev= 30
  4190.0 1749.44  4216.0 1748.57  4306.6 1738.87  4421.8 1724.09  4476.1 1710.86
  4498.0 1708.38  4519.9 1703.71  4579.5 1696.72  4623.7 1686.89  4659.0 1682.32
  4695.1 1672.70  4727.5 1666.53  4777.0 1661.27  4842.7 1661.09  4880.8 1657.66
  4962.8 1657.57  4974.9 1654.92  4975.4 1654.42  4994.5 1654.92  5020.2 1659.36
  5041.3 1660.62  5181.4 1660.38  5228.8 1660.40  5423.9 1660.45  5543.4 1662.88
  5600.0 1673.80  5677.9 1685.42  5755.6 1700.40  5847.7 1708.80  5882.5 1714.34
#Mann=7,-1,0
  4190.0    0.07       0  4727.5   0.035       0  4974.9   0.035       0
  4994.5   0.035       0  5181.4    0.07       0  5228.8   0.035       0
  5423.9    0.07       0
Bank Sta=4974.9,4994.5
Exp/Cntr=0.3,0.1

Type RM Length L Ch R = 1,41491,577,577,577
BEGIN DESCRIPTION:
Mapping XS a1b63e1f
END DESCRIPTION:
XS GIS Cut Line= 3
      1663631.02      6977710.82      1664252.52      6977790.68
      1665300.54      6978144.65
#Sta/Elev= 30
  4377.1 1747.06  4428.4 1743.74  4481.9 1741.67  4612.4 1725.73  4683.6 1705.72
  4708.4 1701.71  4713.8 1699.42  4814.7 1684.94  4867.5 1679.78  4895.3 1671.52
  4919.9 1667.37  4942.1 1659.65  4965.9 1655.30  4996.1 1652.97  5001.4 1650.76
  5001.9 1650.26  5021.1 1650.76  5027.4 1655.00  5059.1 1658.58  5383.5 1657.20
  5451.7 1654.57  5571.6 1655.53  5660.7 1659.78  5724.1 1667.76  5734.8 1670.80
  5823.9 1682.97  5881.5 1695.15  5998.5 1707.54  6038.8 1713.73  6109.9 1718.18
#Mann=7,-1,0
  4377.1   0.035       0  4428.4    0.07       0  4612.4    0.16       0
  4919.9    0.07       0  5001.4    0.07       0  5021.1    0.07       0
  5571.6    0.07       0
Bank Sta=5001.4,5021.1
Exp/Cntr=0.3,0.1

Type RM Length L Ch R = 1,40914,1208,1208,1208
BEGIN DESCRIPTION:
Mapping XS 8798a50d
END DESCRIPTION:
XS GIS Cut Line= 3
      1663706.49      6978326.56      1664105.76      6978319.62
      1665170.87      6978364.72
#Sta/Elev= 30
  4601.5 1731.23  4613.4 1729.74  4700.0 1717.35  4730.0 1710.52  4770.0 1698.89
  4805.7 1691.36  4890.1 1677.41  4950.1 1660.98  4980.1 1655.01  5003.0 1652.38
  5010.1 1648.49  5010.2 1647.31  5010.7 1646.81  5029.9 1647.31  5030.1 1650.85
  5040.1 1655.40  5050.1 1656.67  5103.4 1655.92  5180.2 1653.69  5260.3 1655.24
  5410.4 1650.21  5461.5 1652.96  5540.6 1650.71  5554.5 1652.01  5570.6 1657.25
  5590.6 1659.08  5660.7 1671.16  5850.8 1685.97  5900.9 1693.38  6066.9 1707.82
#Mann=6,-1,0
  4601.5    0.16       0  4613.4    0.07       0  5010.2    0.07       0
  5029.9    0.07       0  5103.4   0.035       0  5461.5    0.07       0
Bank Sta=5010.2,5029.9
Exp/Cntr=0.3,0.1

Type RM Length L Ch R = 1,39706,561,561,561
BEGIN DESCRIPTION:
Mapping XS 4a67ac03
END DESCRIPTION:
XS GIS Cut Line= 3
      1663817.55      6979014.06      1664546.73      6978739.76
      1665240.31      6978483.13
#Sta/Elev= 30
  4212.1 1732.96  4244.3 1730.90  4330.5 1717.09  4380.3 1702.00  4385.6 1701.83
  4391.0 1698.42  4410.5 1692.98  4526.0 1670.56  4556.3 1666.62  4561.9 1663.22
  4581.2 1657.06  4604.7 1654.50  4690.5 1653.91  4812.3 1654.01  4935.3 1651.28
  4977.7 1643.09  4978.2 1642.59  4997.5 1643.09  5032.0 1649.35  5038.4 1652.92
  5043.7 1652.47  5063.4 1659.68  5085.3 1662.65  5170.6 1669.52  5394.5 1681.84
  5552.5 1698.23  5644.8 1705.22  5700.3 1712.23  5728.7 1713.35  5730.7 1713.46
#Mann=8,-1,0
  4212.1    0.16       0  4244.3    0.07       0  4690.5   0.035       0
  4935.3    0.07       0  4977.7    0.07       0  4997.5    0.07       0
  5552.5    0.16       0  5728.7    0.07       0
Bank Sta=4977.7,4997.5
Exp/Cntr=0.3,0.1

Type RM Length L Ch R = 1,39145,444,444,444
BEGIN DESCRIPTION:
Mapping XS b0b92525
END DESCRIPTION:
XS GIS Cut Line= 3
      1663946.06      6979486.28      1664553.67      6979298.78
      1665515.46      6978625.18
#Sta/Elev= 30
  4362.5 1728.62  4370.3 1728.01  4408.0 1725.42  4440.7 1718.52  4528.8 1709.01
  4609.2 1691.23  4738.1 1673.07  4769.5 1667.01  4790.5 1658.63  4826.9 1648.53
  4895.1 1649.49  4946.2 1646.25  4989.3 1646.91  4996.5 1644.49  5026.7 1643.20
  5027.2 1642.70  5046.5 1643.20  5048.5 1643.90  5057.9 1647.85  5085.5 1651.00
  5230.5 1653.39  5307.6 1657.78  5310.9 1658.07  5438.8 1666.06  5459.8 1669.19
  5703.9 1682.98  5786.5 1692.85  6025.6 1712.95  6067.4 1714.85  6172.6 1719.92
#Mann=10,-1,0
  4362.5    0.16       0  4370.3    0.07       0  4826.9   0.035       0
  5026.7   0.035       0  5046.5   0.035       0  5048.5    0.07       0
  5307.6   0.035       0  5310.9    0.07       0  5786.5    0.16       0
  6067.4    0.07       0
Bank Sta=5026.7,5046.5
Exp/Cntr=0.3,0.1

Type RM Length L Ch R = 1,38701,418,418,418
BEGIN DESCRIPTION:
Mapping XS 703a3413
END DESCRIPTION:
XS GIS Cut Line= 3
      1664201.22      6979949.41      1664630.93      6979712.41
      1665589.27      6978915.53
#Sta/Elev= 30
  4510.1 1707.42  4565.3 1707.04  4654.6 1698.67  4690.2 1694.69  4706.3 1690.84
  4793.4 1682.05  4874.8 1667.18  4896.5 1665.28  4925.5 1658.64  4956.1 1643.00
  4961.3 1641.81  4961.8 1641.31  4981.2 1641.81  4983.6 1642.82  5034.9 1643.46
  5063.6 1646.77  5106.1 1648.07  5106.4 1648.06  5204.0 1648.97  5396.9 1651.07
  5527.2 1654.96  5688.5 1662.08  5830.4 1670.23  5922.9 1677.92  5937.2 1680.73
  5972.3 1684.29  6013.8 1691.64  6072.6 1698.45  6192.4 1708.28  6247.2 1714.13
#Mann=9,-1,0
  4510.1    0.16       0  4654.6    0.07       0  4961.3    0.07       0
  4981.2    0.07       0  5106.1   0.035       0  5106.4    0.07       0
  5204.0   0.035       0  5527.2    0.07       0  6013.8    0.16       0
Bank Sta=4961.3,4981.2
Exp/Cntr=0.3,0.1

Type RM Length L Ch R = 1,38283,361,361,361
BEGIN DESCRIPTION:
Mapping XS f4abe965
END DESCRIPTION:
XS GIS Cut Line= 3
      1664505.93      6980355.64      1664821.04      6980063.97
      1665854.54      6979022.66
#Sta/Elev= 30
  4563.7 1704.82  4596.8 1703.60  4702.8 1690.78  4766.8 1685.81  4787.8 1682.99
  4837.2 1675.89  4858.7 1670.58  4908.0 1661.19  4943.7 1651.12  4954.8 1649.24
  4978.9 1642.79  4985.7 1642.32  4990.2 1638.25  4990.7 1637.75  5010.1 1638.25
  5014.3 1640.46  5021.3 1641.94  5035.4 1643.08  5063.7 1642.71  5141.5 1646.50
  5551.6 1648.85  5736.8 1653.43  5777.9 1655.37  5898.1 1668.37  6004.2 1674.34
  6104.1 1684.08  6177.7 1693.43  6265.8 1700.71  6287.0 1700.70  6460.2 1710.06
#Mann=7,-1,0
  4563.7    0.07       0  4954.8   0.035       0  4990.2   0.035       0
  5010.1   0.035       0  5736.8    0.07       0  6104.1    0.16       0
  6177.7    0.07       0
Bank Sta=4990.2,5010.1
Exp/Cntr=0.3,0.1

Type RM Length L Ch R = 1,37922,273,273,273
BEGIN DESCRIPTION:
Mapping XS 173768b2
END DESCRIPTION:
XS GIS Cut Line= 3
      1664787.21      6980506.66      1665091.87      6980274.91
      1666076.27      6979079.56
#Sta/Elev= 30
  4616.9 1692.85  4721.5 1682.21  4777.7 1674.39  4835.8 1660.65  4864.9 1651.54
  4892.0 1645.88  4960.2 1643.17  4985.5 1641.17  4998.5 1642.26  5013.8 1637.84
  5024.7 1637.69  5025.2 1637.19  5044.6 1637.69  5049.0 1641.00  5092.0 1645.47
  5354.8 1646.43  5422.3 1646.64  5651.5 1649.80  5830.9 1654.88  5909.0 1662.67
  5944.2 1664.41  5952.1 1666.53  5972.9 1666.28  6001.6 1669.45  6114.9 1673.50
  6207.5 1679.25  6257.0 1679.83  6320.8 1687.20  6384.7 1697.94  6548.2 1714.27
#Mann=7,-1,0
  4616.9    0.07       0  4960.2   0.035       0  5024.7   0.035       0
  5044.6   0.035       0  5354.8    0.07       0  5422.3   0.035       0
  5651.5    0.07       0
Bank Sta=5024.7,5044.6
Exp/Cntr=0.3,0.1

Type RM Length L Ch R = 1,37649,376,376,376
BEGIN DESCRIPTION:
Mapping XS 2becb8bd
END DESCRIPTION:
XS GIS Cut Line= 3
      1665057.56      6980562.90      1665297.16      6980443.10
      1666174.79      6979219.11
#Sta/Elev= 30
  4722.6 1675.15  4763.0 1668.00  4807.7 1658.23  4820.4 1653.36  4842.7 1648.10
  4865.1 1644.50  4896.1 1643.35  4941.9 1640.79  4993.0 1640.22  4997.8 1635.94
  4998.3 1635.44  5017.7 1635.94  5028.6 1641.78  5058.1 1644.69  5226.2 1644.63
  5320.5 1644.98  5538.2 1647.35  5772.9 1652.98  5887.2 1657.09  5942.8 1659.60
  6009.9 1662.57  6066.2 1666.80  6104.2 1669.72  6282.5 1679.41  6353.8 1687.37
  6383.2 1693.38  6411.8 1697.36  6425.0 1698.08  6433.6 1699.92  6496.6 1704.49
#Mann=9,-1,0
  4722.6    0.07       0  4896.1   0.035       0  4997.8   0.035       0
  5017.7   0.035       0  5226.2    0.07       0  5320.5   0.035       0
  5887.2    0.07       0  5942.8   0.035       0  6066.2    0.07       0
Bank Sta=4997.8,5017.7
Exp/Cntr=0.3,0.1

Type RM Length L Ch R = 1,37273,306,306,306
BEGIN DESCRIPTION:
Swager Creek 62.0
END DESCRIPTION:
XS GIS Cut Line= 3
      1665355.04      6980737.98      1665605.00      6980638.00
      1666385.70      6979128.00
#Sta/Elev= 30
  4730.3 1658.76  4751.8 1656.25  4762.6 1655.25  4774.7 1651.38  4793.5 1648.34
  4805.7 1643.88  4828.5 1640.41  4924.1 1641.28  4978.0 1640.11  4984.7 1639.40
  4986.9 1637.46  4987.4 1636.96  5006.8 1637.46  5029.9 1638.47  5035.5 1641.60
  5067.1 1643.82  5273.5 1643.25  5400.7 1644.65  5812.1 1653.20  5993.0 1658.98
  6119.5 1668.22  6133.8 1669.23  6363.8 1680.71  6452.4 1689.02  6468.9 1692.74
  6507.6 1696.19  6579.7 1698.87  6586.8 1700.45  6618.3 1702.18  6699.4 1703.96
#Mann=7,-1,0
  4730.3    0.07       0  4751.8   0.035       0  4986.9   0.035       0
  5006.8   0.035       0  5812.1    0.07       0  6119.5   0.035       0
  6133.8    0.07       0
Bank Sta=4986.9,5006.8
Exp/Cntr=0.3,0.1

Type RM Length L Ch R = 1,36967,1080,1080,1080
BEGIN DESCRIPTION:
Mapping XS 8aba9dcb
END DESCRIPTION:
XS GIS Cut Line= 3
      1665195.53      6980845.42      1665718.56      6980901.24
      1667425.17      6979201.72
#Sta/Elev= 30
  4474.0 1664.76  4624.3 1657.85  4714.8 1655.70  4765.1 1651.39  4815.4 1643.74
  4849.4 1642.42  4966.4 1636.25  4966.9 1635.75  4986.3 1636.25  5070.5 1642.69
  5374.5 1641.08  6053.2 1649.64  6082.9 1650.19  6279.6 1652.71  6316.9 1649.43
  6365.2 1651.56  6392.8 1653.99  6477.6 1654.71  6534.2 1653.85  6541.3 1652.40
  6548.3 1654.00  6555.4 1652.71  6661.5 1658.04  7049.0 1666.55  7099.9 1669.36
  7206.0 1679.40  7261.8 1681.72  7368.7 1684.85  7372.7 1685.15  7408.5 1686.43
#Mann=12,-1,0
  4474.0    0.07       0  4849.4   0.035       0  4966.4   0.035       0
  4986.3   0.035       0  6053.2    0.07       0  6082.9   0.035       0
  6316.9    0.07       0  6365.2   0.035       0  7049.0    0.07       0
  7261.8   0.035       0  7368.7    0.07       0  7372.7   0.035       0
Bank Sta=4966.4,4986.3
Exp/Cntr=0.3,0.1

Type RM Length L Ch R = 1,35887,613,613,613
BEGIN DESCRIPTION:
Mapping XS 0513d031
END DESCRIPTION:
XS GIS Cut Line= 3
      1665273.70      6980945.26      1666558.38      6981342.38
      1667270.08      6980359.45
#Sta/Elev= 30
  3654.3 1653.71  3739.4 1650.45  3811.7 1645.96  3816.9 1644.20  3823.1 1643.63
  3854.8 1642.29  3958.8 1641.74  3962.5 1641.84  4173.4 1642.16  4576.7 1641.42
  4744.7 1638.62  4762.0 1638.06  4767.2 1640.08  4781.1 1639.90  4838.4 1640.14
  4932.9 1633.69  4933.4 1633.19  4953.3 1633.69  4968.2 1634.88  5014.7 1634.45
  5029.1 1637.48  5041.7 1638.49  5150.8 1638.32  5260.0 1641.72  5392.3 1644.28
  5522.9 1645.58  5841.1 1651.90  5949.9 1654.50  6030.3 1656.68  6212.5 1662.18
#Mann=13,-1,0
  3654.3    0.07       0  3958.8   0.035       0  3962.5    0.07       0
  4173.4   0.035       0  4744.7    0.07       0  4781.1   0.035       0
  4932.9   0.035       0  4953.3   0.035       0  5260.0    0.07       0
  5392.3   0.035       0  5841.1    0.07       0  5949.9   0.035       0
  6030.3    0.07       0
Bank Sta=4932.9,4953.3
Exp/Cntr=0.3,0.1

Type RM Length L Ch R = 1,35274,685,685,685
BEGIN DESCRIPTION:
Swager Creek 60.0
END DESCRIPTION:
XS GIS Cut Line= 3
      1665091.35      6980884.47      1666225.06      6981688.20
      1666342.80      6982684.27
#Sta/Elev= 30
  3610.3 1662.25  3658.7 1660.03  3694.3 1655.04  3759.6 1652.67  3872.7 1644.00
  3928.8 1641.77  4235.2 1639.95  4258.8 1639.88  4433.8 1639.40  4475.6 1637.44
  4692.2 1638.08  4742.5 1636.27  4935.8 1632.77  4942.0 1629.96  4965.3 1628.35
  4965.8 1627.85  4989.9 1628.35  4992.4 1630.60  5002.4 1629.58  5010.4 1635.96
  5250.7 1643.24  5349.5 1646.69  5422.7 1650.01  5555.9 1658.35  5638.8 1667.30
  5674.5 1675.20  5721.7 1681.56  5825.5 1690.87  5875.9 1698.09  6003.0 1707.47
#Mann=11,-1,0
  3610.3    0.07       0  3928.8   0.035       0  4235.2    0.07       0
  4258.8   0.035       0  4742.5    0.07       0  4965.3    0.07       0
  4989.9    0.07       0  5010.4   0.035       0  5250.7    0.07       0
  5349.5   0.035       0  5422.7    0.07       0
Bank Sta=4965.3,4989.9
Exp/Cntr=0.3,0.1
