--- Deadman 02.prj (project) ---

Proj Title=Deadman 02 Base Level Engineering
Current Plan=p01
Default Exp/Contr=0.3,0.1
English Units
Geom File=g01
Flow File=f01
Plan File=p01
Y Axis Title=Elevation
X Axis Title(PF)=Main Channel Distance
X Axis Title(XS)=Station
BEGIN DESCRIPTION:
Deadman 02
END DESCRIPTION:
DSS Export Rating Curves= 0
DSS Export Rating Curve Sorted= 0
DSS Export Volume Flow Curves= 0
DXF OffsetX= 0
DXF OffsetY= 0
DXF ScaleX= 1
DXF ScaleY= 10

--- Deadman 02.p01 (plan) ---

Plan Title=Multiple Run
Short Identifier=Multiple
Geom File=g01
Flow File=f01
Subcritical Flow
K Sum by GR= 0
Std Step Tol= 0.01
Critical Tol= 0.01
Num of Std Step Trials= 20
Max Error Tol= 0.3
Flow Tol Ratio= 0.001
Split Flow NTrial= 30
Split Flow Tol= 0.02
Split Flow Ratio= 0.02
Log Output Level= 0
Friction Slope Method= 1
Unsteady Friction Slope Method= 2
Unsteady Bridges Friction Slope Method= 1
Parabolic Critical Depth
Global Vel Dist=  1 , 1 , 1
Global Log Level= 0
CheckData=True
Encroach Param= -1, 0, 0, 0
BEGIN DESCRIPTION:
Multiple Run
END DESCRIPTION:

--- Deadman 02.f01 (steady flow) ---

Flow Title=Multiple
Number of Profiles=7
Profile Names=10-year,25-year,50-year,1pct_min,100-year,1pct_plu,500-year
River Rch & RM= Deadman 02,Reach-1,39303
     327     453     556     340     678    1353    1020
River Rch & RM= Deadman 02,Reach-1,28028
     408     573     711     438     874    1744    1339
River Rch & RM= Deadman 02,Reach-1,26082
     485     687     857     532    1061    2116    1645
River Rch & RM= Deadman 02,Reach-1,21926
     552     787     986     613    1224    2442    1911
River Rch & RM= Deadman 02,Reach-1,18269
     583     833    1045     651    1298    2591    2033
River Rch & RM= Deadman 02,Reach-1,17163
     763    1103    1396     877    1749    3490    2782
River Rch & RM= Deadman 02,Reach-1,12807
     831    1206    1530     962    1919    3830    3063
River Rch & RM= Deadman 02,Reach-1,9403
     889    1293    1642    1034    2063    4117    3302
River Rch & RM= Deadman 02,Reach-1,2954
     900    1308    1661    1046    2086    4163    3336
Boundary for River Rch & Prof#=Deadman 02,Reach-1,1
Up Type=0
Dn Type=3
Dn Slope=0.009
Boundary for River Rch & Prof#=Deadman 02,Reach-1,2
Up Type=0
Dn Type=3
Dn Slope=0.009
Boundary for River Rch & Prof#=Deadman 02,Reach-1,3
Up Type=0
Dn Type=3
Dn Slope=0.009
Boundary for River Rch & Prof#=Deadman 02,Reach-1,4
Up Type=0
Dn Type=3
Dn Slope=0.009
Boundary for River Rch & Prof#=Deadman 02,Reach-1,5
Up Type=0
Dn Type=3
Dn Slope=0.009
Boundary for River Rch & Prof#=Deadman 02,Reach-1,6
Up Type=0
Dn Type=3
Dn Slope=0.009
Boundary for River Rch & Prof#=Deadman 02,Reach-1,7
Up Type=0
Dn Type=3
Dn Slope=0.009

--- Deadman 02.g01 (geometry) ---

Geom Title=Existing Conditions
Program Version=4.10

River Reach=Deadman 02      ,Reach-1
Reach XY= 30
        1588755.        6944188.      1589652.26      6945132.66
       1590614.8      6945148.48      1591352.55      6946182.53
      1592353.42      6946241.83      1593811.19      6947145.82
      1594752.55      6948532.54      1598430.18      6948037.54
      1599643.28      6948236.95        1600253.      6947582.31
      1600008.46      6946795.74      1600425.17      6946868.44
      1601100.03      6945790.58      1601760.44      6942943.25
      1603363.48      6941491.51      1605264.66      6940727.83
      1605348.86      6940145.73      1606068.83      6940074.67
      1605841.26      6939501.19      1606749.37      6939586.39
      1607049.99      6939187.12      1607694.36      6939487.45
      1608079.88      6939087.68      1608958.29      6939329.95
      1610025.21      6938637.63      1611015.49      6939487.07
      1611110.45      6938990.05      1611757.74      6938993.34
      1612174.99      6939538.07        1612505.        6939088.

Type RM Length L Ch R = 1 ,39303   ,775,775,775
BEGIN DESCRIPTION:
Deadman 02 66.0
END DESCRIPTION:
XS GIS Cut Line= 3
      1588555.01      6944937.96      1588802.31      6944234.78
      1589079.33      6943384.89
#Sta/Elev= 30
  4254.6 1725.79  4264.7 1725.39  4275.8 1722.32  4318.2 1720.63  4326.7 1721.06
  4357.7  1718.6  4371.2 1719.65  4381.8 1719.51  4393.9 1717.38  4419.6 1716.41
    4456 1713.36  4507.2 1712.81  4512.5 1713.64  4538.2 1710.22  4583.2 1708.29
  4731.6 1706.37  5122.6 1706.02  5122.9 1705.52  5127.2 1706.02  5364.7 1706.37
    5513 1708.45    5545 1709.47  5554.1 1710.42  5571.6 1715.46  5596.1 1716.67
  5617.2 1714.23  5635.4 1715.37  5640.7 1714.77  5763.1 1717.99  5893.9 1716.69
#Mann= 3 ,-1 , 0
  4254.6     .05       0  5122.6    .035       0  5127.2     .05       0
Bank Sta=5122.6,5127.2
XS Rating Curve= 0 ,0
Exp/Cntr=0.3,0.1

Type RM Length L Ch R = 1 ,38528   ,479,479,479
BEGIN DESCRIPTION:
Deadman 02 65.0
END DESCRIPTION:
XS GIS Cut Line= 3
      1588654.99      6945338.01        1589405.        6944688.
      1590580.03      6944212.99
#Sta/Elev= 30
  4007.4 1730.73  4021.2 1728.94    4043 1722.77  4071.5 1720.37    4326 1717.76
  4397.3 1718.27  4446.7 1716.87  4489.4 1713.69  4602.9 1709.15  4695.5 1706.78
  4730.7 1707.17  4759.2 1705.63    4780 1707.83  4815.1 1705.51  4891.7 1705.06
  4892.1 1704.56  4896.3 1705.06  5215.6 1705.34  5551.1 1708.48  5623.5 1712.17
  5647.1 1711.65  5682.5 1712.99  5730.8 1716.65  5765.7  1715.7  5784.4 1716.91
  5927.5  1716.8  6082.2 1722.76  6121.7 1724.85  6130.5 1726.51  6267.3 1726.33
#Mann= 3 ,-1 , 0
  4007.4     .05       0  4891.7     .05       0  4896.3     .05       0
Bank Sta=4891.7,4896.3
XS Rating Curve= 0 ,0
Exp/Cntr=0.3,0.1

Type RM Length L Ch R = 1 ,38049   ,655,655,655
BEGIN DESCRIPTION:
Deadman 02 64.0
END DESCRIPTION:
XS GIS Cut Line= 3
      1588955.02      6945637.98        1589605.        6945088.
      1590205.04      6944737.98
#Sta/Elev= 30
  4143.9 1720.91  4208.2 1718.95  4249.9 1720.26  4271.9 1718.21  4392.8 1714.43
  4456.5 1713.56  4520.2 1715.14  4654.7 1711.28  4797.1 1710.13  4803.6 1708.55
  4832.2 1709.93  4895.9 1708.12  4914.4 1704.71  4914.7 1704.21  4919.1 1704.71
  4924.5 1708.65    4931 1708.76  4967.4 1707.91  4988.2 1705.31  5067.7    1708
  5147.9 1706.09  5163.6 1708.06  5200.8 1709.15  5286.8 1708.21  5382.8 1711.64
    5463 1712.39  5580.4 1718.59  5600.6 1718.34  5672.5 1723.65    5690 1724.04
#Mann= 5 ,-1 , 0
  4143.9     .05       0  4914.4     .05       0  4919.1     .05       0
  5600.6     .12       0  5672.5     .05       0
Bank Sta=4914.4,4919.1
XS Rating Curve= 0 ,0
Exp/Cntr=0.3,0.1

Type RM Length L Ch R = 1 ,37394   ,283,283,283
BEGIN DESCRIPTION:
Mapping XS c256b9d4
END DESCRIPTION:
XS GIS Cut Line= 3
      1590292.62      6946550.92      1590214.38      6946217.38
      1590251.19      6944778.14
#Sta/Elev= 30
  3577.6 1720.07  3621.7 1719.89  3629.8 1721.38  3642.2 1720.44  3652.5 1718.28
  3755.2 1718.69  3908.1 1716.56  4075.9 1716.97  4219.7 1717.64  4259.7 1718.55
  4329.7 1716.93  4369.7 1717.62  4459.7 1716.52  4509.8 1716.92  4532.9 1717.94
  4559.8 1714.83  4619.8 1715.78  4809.9 1713.47  4949.9  1713.6  5017.4 1712.68
  5017.8 1712.18  5022.5 1712.68  5069.9 1715.68    5090 1715.13    5140 1715.77
    5190 1717.32  5287.8 1719.51    5320 1721.58    5340 1721.71  5359.9 1723.68
#Mann= 7 ,-1 , 0
  3577.6     .05       0  3908.1     .12       0  4075.9     .05       0
  5017.4     .05       0  5022.5     .05       0    5190     .12       0
  5287.8     .05       0
Bank Sta=5017.4,5022.5
XS Rating Curve= 0 ,0
Exp/Cntr=0.3,0.1

Type RM Length L Ch R = 1 ,37111   ,174,174,174
BEGIN DESCRIPTION:
Mapping XS b4bec68e
END DESCRIPTION:
XS GIS Cut Line= 2
      1590503.18      6945472.29       1590558.7      6944632.52
#Sta/Elev= 30
  4664.6 1721.54    4719 1720.03  4749.1 1720.82    4766 1720.56  4771.1 1719.75
  4779.1 1720.04  4809.2 1718.79  4839.3 1715.74  4899.4 1712.24    4917 1712.25
    4922 1713.06    4947 1711.96  4947.4 1711.46  4951.7 1711.46  4952.1 1711.96
  4979.6 1713.61  4989.6 1712.95  5009.6 1713.65  5029.7 1713.46  5049.7 1715.18
  5089.8  1713.8  5107.2 1714.08  5237.4 1717.59  5280.2 1720.02  5374.9  1721.6
  5400.5 1722.87  5460.6 1723.31  5480.7 1725.55  5500.7 1725.09  5506.2 1724.31
#Mann= 5 ,-1 , 0
  4664.6     .05       0    4947     .05       0  4952.1     .05       0
  5107.2     .12       0  5237.4     .05       0
Bank Sta=4947,4952.1
XS Rating Curve= 0 ,0
Exp/Cntr=0.3,0.1

Type RM Length L Ch R = 1 ,36937   ,299,299,299
BEGIN DESCRIPTION:
Mapping XS 248ccfc3
END DESCRIPTION:
XS GIS Cut Line= 2
       1590511.6      6945524.69      1590993.38      6944578.49
#Sta/Elev= 30
  4643.2 1723.02  4650.7 1723.35    4659 1721.61  4664.6 1722.56  4681.3 1721.84
  4709.1 1719.19  4731.4 1719.55  4753.6 1717.78  4770.2 1717.78  4820.3 1714.08
  4859.2 1713.03  4897.6 1713.65  4909.3 1711.53  4931.5 1710.17  5034.6 1708.56
    5035 1708.06  5039.7 1708.56  5155.7  1709.6  5365.1 1715.68  5387.4 1716.93
  5402.6 1719.53    5425 1721.33  5473.8 1723.24  5517.8 1725.88  5559.7 1727.54
  5609.8 1731.48  5648.6 1731.93  5683.1 1734.06  5698.7  1734.2    5705 1733.28
#Mann= 5 ,-1 , 0
  4643.2     .05       0  5034.6     .05       0  5039.7     .05       0
  5473.8     .12       0  5517.8     .05       0
Bank Sta=5034.6,5039.7
XS Rating Curve= 0 ,0
Exp/Cntr=0.3,0.1

Type RM Length L Ch R = 1 ,36638   ,440,440,440
BEGIN DESCRIPTION:
Deadman 02 61.0
END DESCRIPTION:
XS GIS Cut Line= 3
      1590505.04      6945537.99        1590855.        6945438.
      1591255.02      6945087.98
#Sta/Elev= 30
  4641.5 1723.24  4672.7 1722.34  4692.2 1720.59  4697.4 1721.07  4714.3 1718.93
  4745.5 1717.23  4776.7 1717.63  4787.1  1715.4    4804 1713.26  4849.5 1708.73
  4901.5 1705.43  4961.3 1704.08  4961.7 1703.58  4966.4 1704.08  5026.8 1704.74
  5051.3 1705.76  5098.2 1705.78  5133.1 1707.01  5161.6 1707.03  5191.7 1708.47
  5218.1 1710.48  5225.2 1711.68  5246.1 1712.28  5267.9 1714.09  5336.4 1717.76
  5352.4 1718.12  5430.7 1722.67  5466.3 1725.98  5494.7 1727.45    5537 1731.66
#Mann= 7 ,-1 , 0
  4641.5     .05       0  4961.3     .05       0  4966.4     .05       0
  5051.3     .12       0  5098.2     .05       0  5191.7     .12       0
  5336.4     .05       0
Bank Sta=4961.3,4966.4
XS Rating Curve= 0 ,0
Exp/Cntr=0.3,0.1

Type RM Length L Ch R = 1 ,36198   ,441,441,441
BEGIN DESCRIPTION:
Deadman 02 60.0
END DESCRIPTION:
XS GIS Cut Line= 3
      1590654.97        6945788.        1591005.        6945838.
      1591405.02      6945437.98
#Sta/Elev= 30
  4637.7 1718.81    4668 1717.24  4688.2 1714.91  4698.3 1714.59  4708.4 1712.96
  4738.7 1709.98  4809.5 1704.37  4839.8 1702.87  4890.3 1702.51  4948.3 1700.06
  4948.7 1699.56  4953.1 1699.56  4953.5 1700.06  4981.2 1700.73  5005.4 1700.26
  5033.7 1701.18  5076.1 1700.81  5104.4 1701.96  5146.9 1701.88  5175.1 1702.91
  5203.4 1704.75  5231.7 1705.25  5245.8 1706.81  5274.1 1707.51  5316.6 1710.31
  5348.9 1711.61  5490.9 1721.72  5500.4  1722.7  5528.7 1723.82    5557 1725.79
#Mann= 5 ,-1 , 0
  4637.7     .05       0  4948.3     .03       0  4953.5     .05       0
  5348.9     .12       0  5490.9     .05       0
Bank Sta=4948.3,4953.5
XS Rating Curve= 0 ,0
Exp/Cntr=0.3,0.1

Type RM Length L Ch R = 1 ,35757   ,587,587,587
BEGIN DESCRIPTION:
Deadman 02 59.0
END DESCRIPTION:
XS GIS Cut Line= 3
      1590704.99        6946438.        1591305.        6946138.
      1591704.99      6945738.01
#Sta/Elev= 30
  4329.6 1725.55  4334.9 1725.71  4360.4 1724.04  4382.7 1721.58  4410.7 1720.54
  4477.8 1716.28  4486.1 1715.02  4522.5 1711.95  4530.9 1710.09  4553.2 1708.68
  4620.3 1706.31    4665 1703.49  4718.1 1702.67  4740.5 1703.39  4762.8 1701.11
  4799.2 1700.57  4813.2 1700.85  4821.5 1701.84  4843.9 1700.99    4995 1700.13
  4995.4 1699.63  4999.8 1699.63  5000.2 1700.13  5127.7 1700.82  5269.1 1704.23
  5325.7 1706.29    5453 1712.42  5509.5 1712.59  5537.8 1713.97  5566.1 1716.28
#Mann= 4 ,-1 , 0
  4329.6     .12       0  4334.9     .05       0    4995     .05       0
  5000.2     .05       0
Bank Sta=4995,5000.2
XS Rating Curve= 0 ,0
Exp/Cntr=0.3,0.1

Type RM Length L Ch R = 1 ,35170   ,313,313,313
BEGIN DESCRIPTION:
Deadman 02 58.0
END DESCRIPTION:
XS GIS Cut Line= 3
      1591969.04      6947150.16      1591857.51      6946238.15
        1591955.      6945937.99
#Sta/Elev= 30
  4081.2 1709.03  4157.3  1708.4    4174 1709.28  4204.3 1709.68  4264.7 1707.41
  4315.1 1706.82  4335.2 1705.75  4395.7 1706.74  4446.1 1705.73  4564.8 1706.39
  4617.3 1704.89  4667.7 1705.06  4697.9  1703.8  4748.3 1702.83  4957.2 1700.99
  4957.6 1700.49  4962.2 1700.49  4962.6 1700.99  5075.9 1701.36  5139.8 1703.78
  5157.9 1705.44  5198.5 1707.77  5210.4 1709.86  5230.4 1711.01  5235.7 1712.96
  5262.4  1714.6  5267.6 1716.48  5294.3 1718.82  5299.6  1720.2  5315.6 1720.45
#Mann= 3 ,-1 , 0
  4081.2     .05       0  4957.2     .03       0  4962.6     .05       0
Bank Sta=4957.2,4962.6
XS Rating Curve= 0 ,0
Exp/Cntr=0.3,0.1

Type RM Length L Ch R = 1 ,34857   ,442,442,442
BEGIN DESCRIPTION:
Deadman 02 57.0
END DESCRIPTION:
XS GIS Cut Line= 3
        1592205.        6946538.        1592155.        6946188.
        1592105.      6945938.01
#Sta/Elev= 30
  4650.8 1718.67    4671 1718.36  4681.1 1717.89  4691.2 1717.04  4701.3 1717.06
  4731.6 1715.66  4782.1 1712.12  4802.3 1711.42  4883.1 1705.64  4943.7 1702.52
  4974.1 1702.78  4991.6 1701.97    4992 1701.47  4996.6 1701.47    4997 1701.97
  5001.8 1703.06  5024.8 1703.84  5045.2 1705.41  5065.5  1705.6  5075.7 1706.25
  5096.1 1708.21  5106.3 1708.59  5126.7 1710.12  5167.5 1713.87  5177.7 1713.76
  5208.3 1715.29  5218.5 1715.43  5238.9 1716.83  5249.1 1718.41  5259.3 1718.78
#Mann= 3 ,-1 , 0
  4650.8     .05       0  4991.6     .03       0    4997     .05       0
Bank Sta=4991.6,4997
XS Rating Curve= 0 ,0
Exp/Cntr=0.3,0.1

Type RM Length L Ch R = 1 ,34415   ,338,338,338
BEGIN DESCRIPTION:
Deadman 02 56.0
END DESCRIPTION:
XS GIS Cut Line= 3
      1592354.99      6946488.01        1592555.        6946338.
        1592455.      6945638.02
#Sta/Elev= 30
  4755.9 1717.04  4777.8 1715.43    4784 1713.31  4792.4 1713.13  4798.6 1711.38
  4827.8  1710.4  4848.6 1708.42  4877.8  1706.6    4884 1705.18  4919.5    1702
  4948.6 1700.01  5000.1 1698.21  5000.5 1697.71  5005.1 1697.71  5005.5 1698.21
  5066.5 1698.81  5086.7 1699.82  5137.2 1700.43  5147.3 1701.46  5228.1  1703.3
    5309  1704.1  5440.3 1706.62  5460.5 1707.84  5521.1  1710.1  5536.2 1710.09
  5571.6 1711.63  5601.9 1711.96  5632.2 1713.35  5672.6 1714.06    5713 1715.84
#Mann= 3 ,-1 , 0
  4755.9     .05       0  5000.1     .05       0  5005.5     .05       0
Bank Sta=5000.1,5005.5
XS Rating Curve= 0 ,0
Exp/Cntr=0.3,0.1

Type RM Length L Ch R = 1 ,34077   ,451,451,451
BEGIN DESCRIPTION:
Mapping XS 37f24bbb
END DESCRIPTION:
XS GIS Cut Line= 2
      1592641.59      6946747.93      1593009.94      6946308.62
#Sta/Elev= 30
  4735.6 1702.71  4745.4 1703.04  4751.9 1702.26  4759.7 1702.52  4766.2 1702.07
    4774 1702.58  4780.5 1701.85  4794.8 1702.47  4823.4 1701.96  4829.9 1701.18
    4852 1701.18    4866 1699.97  4872.9  1699.9  4879.4 1699.04  4887.2 1698.86
  4893.7 1697.28  4936.6  1695.4  4957.5 1695.58    5029 1694.78  5078.4 1695.37
  5086.2 1696.33  5100.5 1695.71  5107.1 1695.99  5111.3 1694.68  5111.7 1694.18
  5116.3 1694.18  5116.7 1694.68  5135.7 1695.93  5164.3  1696.7  5308.9 1697.17
#Mann= 3 ,-1 , 0
  4735.6     .05       0  5111.3     .05       0  5116.7     .05       0
Bank Sta=5111.3,5116.7
XS Rating Curve= 0 ,0
Exp/Cntr=0.3,0.1

Type RM Length L Ch R = 1 ,33626   ,306,306,306
BEGIN DESCRIPTION:
Mapping XS c697f127
END DESCRIPTION:
XS GIS Cut Line= 2
      1592861.23      6947116.35      1593312.77      6946691.77
#Sta/Elev= 30
  4630.9 1695.42  4653.5 1694.45  4660.8 1693.71  4667.7  1693.8    4675 1692.98
  4681.8 1693.18  4689.1 1692.63  4710.2 1692.75  4731.6 1691.99  4752.7 1691.87
    4802 1689.97  4837.6 1689.51  4872.8 1689.79  4922.6 1688.02  4965.1 1687.47
    4972 1687.83  5000.3 1686.42  5011.7 1686.39  5012.1 1685.89  5016.7 1685.89
  5017.2 1686.39  5021.3  1687.4  5028.6 1686.93  5035.5 1687.14  5042.8 1688.06
  5071.1 1687.81  5170.2 1691.43  5205.4 1691.89  5240.6 1691.68  5250.7 1691.19
#Mann= 3 ,-1 , 0
  4630.9     .05       0  5011.7     .05       0  5017.2     .05       0
Bank Sta=5011.7,5017.2
XS Rating Curve= 0 ,0
Exp/Cntr=0.3,0.1

Type RM Length L Ch R = 1 ,33320   ,204,204,204
BEGIN DESCRIPTION:
Mapping XS 921a0297
END DESCRIPTION:
XS GIS Cut Line= 2
      1593239.43       6947307.5       1593477.8      6946814.18
#Sta/Elev= 30
  4712.2 1685.14  4767.2 1684.65  4800.2  1685.4  4811.6 1684.63  4833.9 1684.23
  4879.1 1684.07  4918.7 1684.45  4933.8 1684.16  4963.9 1682.72  5009.1 1682.44
  5011.8 1682.13  5012.3 1681.63  5017.1 1681.63  5017.5 1682.13  5059.9 1682.48
  5076.9 1683.13  5082.5 1682.92  5122.1 1683.78  5150.3 1683.38  5172.9 1685.16
  5178.4 1685.04  5189.2 1685.72  5195.5 1686.42    5201 1686.17  5218.1 1687.48
  5223.6 1687.23  5233.6 1687.66  5240.7 1688.53  5246.2 1688.11  5260.1 1688.61
#Mann= 3 ,-1 , 0
  4712.2     .05       0  5011.8     .05       0  5017.5     .05       0
Bank Sta=5011.8,5017.5
XS Rating Curve= 0 ,0
Exp/Cntr=0.3,0.1

Type RM Length L Ch R = 1 ,33116   ,102,102,102
BEGIN DESCRIPTION:
Mapping XS f9b8d986
END DESCRIPTION:
XS GIS Cut Line= 2
      1593547.56      6947770.36      1593558.41      6946804.62
#Sta/Elev= 30
  4318.6 1683.99    4371 1683.01    4401 1683.17    4421 1681.65    4441 1681.92
    4451 1682.63    4471 1681.33    4491 1680.86    4501 1681.17    4531 1680.38
    4631 1680.59  4678.1 1679.83  4678.6 1679.33  4683.4 1679.33  4683.8 1679.83
    4731 1681.16    4741 1680.28    4811 1681.15    4871 1679.84    4951 1680.34
    4971 1679.92    5061 1680.74    5081 1680.42    5111 1681.78    5121 1681.07
    5141 1681.97    5181 1682.55    5191 1684.01    5201 1684.34  5284.4 1685.42
#Mann= 3 ,-1 , 0
  4318.6     .05       0  4678.1     .05       0  4683.8     .05       0
Bank Sta=4678.1,4683.8
XS Rating Curve= 0 ,0
Exp/Cntr=0.3,0.1

Type RM Length L Ch R = 1 ,33014   ,218,218,218
BEGIN DESCRIPTION:
Mapping XS 7071ff60
END DESCRIPTION:
XS GIS Cut Line= 2
      1593638.57      6947596.24      1593648.71       6946808.8
#Sta/Elev= 30
  4530.2 1680.42  4548.4 1681.18  4558.4 1681.11  4598.4 1680.16  4608.4 1679.69
  4618.4 1679.79  4648.4 1679.31  4658.4 1678.59  4668.4 1678.79  4688.4 1678.08
  4728.5 1677.18  4765.6 1676.94  4766.1 1676.44  4770.9 1676.44  4771.3 1676.94
  4898.5  1677.8  4918.5 1678.56  4928.5 1679.35  4948.5 1680.25  4968.5 1679.22
  4998.5 1679.21  5008.5 1679.48  5038.5 1679.29  5068.5 1679.76  5088.5 1679.78
  5108.5 1680.41  5118.5 1681.12  5128.5 1681.04  5158.5 1682.15  5317.7 1683.94
#Mann= 3 ,-1 , 0
  4530.2     .05       0  4765.6     .03       0  4771.3     .05       0
Bank Sta=4765.6,4771.3
XS Rating Curve= 0 ,0
Exp/Cntr=0.3,0.1

Type RM Length L Ch R = 1 ,32796   ,371,371,371
BEGIN DESCRIPTION:
Mapping XS 163a2bea
END DESCRIPTION:
XS GIS Cut Line= 2
      1593675.76      6947606.34        1594108.      6946512.23
#Sta/Elev= 30
  4540.7 1678.72  4592.7 1678.74  4637.5 1677.43  4678.7 1678.06  4715.9 1676.44
  4796.9 1675.73  4797.4 1675.23  4802.2 1675.23  4802.6 1675.73  4956.7 1677.52
  5010.8 1678.95    5055 1681.21  5076.5 1681.55  5154.1 1681.29  5248.6  1679.7
  5400.2 1681.14  5442.1 1682.11  5454.3 1682.92  5495.9 1683.33  5508.4 1682.89
  5527.4 1683.44  5532.8 1682.43  5557.1 1682.82  5562.5 1682.06  5581.5 1682.35
  5586.9 1681.87  5611.2 1682.72  5616.6 1681.89  5665.3 1684.08  5717.1 1687.58
#Mann= 3 ,-1 , 0
  4540.7     .05       0  4796.9     .03       0  4802.6     .05       0
Bank Sta=4796.9,4802.6
XS Rating Curve= 0 ,0
Exp/Cntr=0.3,0.1

Type RM Length L Ch R = 1 ,32425   ,224,224,224
BEGIN DESCRIPTION:
Mapping XS 794da437
END DESCRIPTION:
XS GIS Cut Line= 3
      1593735.35      6947588.71      1594060.69        6947564.
      1594261.99      6947021.73
#Sta/Elev= 30
  4542.7 1677.42  4572.4 1677.77  4617.8  1677.3  4622.8 1676.71  4702.8 1674.96
  4732.9  1675.3    4783 1673.65  4833.2 1673.58  4926.3 1670.49  4926.8 1669.99
  4931.7 1669.99  4932.2 1670.49    4949 1671.12  4954.3  1670.7    5046 1671.53
  5095.5 1673.79  5150.9 1675.21  5156.2 1674.14    5174 1674.35    5206  1675.9
  5216.9 1677.19  5236.6 1677.28  5248.7 1676.28  5272.3 1675.82  5297.4 1676.75
  5327.7 1676.25  5383.1 1677.02  5430.1 1678.02  5438.5 1678.84  5447.4    1678
#Mann= 3 ,-1 , 0
  4542.7     .05       0  4926.3     .03       0  4932.2     .05       0
Bank Sta=4926.3,4932.2
XS Rating Curve= 0 ,0
Exp/Cntr=0.3,0.1

Type RM Length L Ch R = 1 ,32201   ,154,154,154
BEGIN DESCRIPTION:
Mapping XS 5a0224aa
END DESCRIPTION:
XS GIS Cut Line= 3
      1593719.71      6947602.99      1594317.87      6947599.62
      1594689.65      6947575.96
#Sta/Elev= 30
  4454.8 1677.44  4490.1 1677.84  4590.1  1677.5  4610.1 1676.23  4620.1 1676.15
  4630.1  1675.3  4650.1 1675.23  4670.1 1675.76  4690.1 1674.62  4750.1 1673.43
  4780.1 1673.45  4900.1 1671.41  4990.1 1668.74  5030.1 1669.26  5040.1 1668.83
  5077.2 1668.39  5077.7 1667.89  5082.6 1667.89  5083.1 1668.39  5100.2 1668.82
  5130.3 1668.88  5140.3  1669.4  5161.2 1669.71  5190.4 1669.79  5200.4 1670.25
  5240.5 1670.42  5330.7 1673.89  5340.7 1674.82  5400.8 1675.12  5425.5 1675.78
#Mann= 3 ,-1 , 0
  4454.8     .05       0  5077.2     .03       0  5083.1     .05       0
Bank Sta=5077.2,5083.1
XS Rating Curve= 0 ,0
Exp/Cntr=0.3,0.1

Type RM Length L Ch R = 1 ,32047   ,380,380,380
BEGIN DESCRIPTION:
Mapping XS 2b569f5b
END DESCRIPTION:
XS GIS Cut Line= 2
      1593983.34      6947728.04      1594794.38      6947707.76
#Sta/Elev= 30
  4626.1 1678.04  4657.8 1678.03  4667.8 1677.34  4677.8 1677.25  4697.8 1676.41
  4727.8 1674.21  4737.8 1673.97  4747.8 1674.58  4757.8 1676.02  4777.8 1675.77
  4787.8 1673.63  4807.8 1671.11  4837.8 1670.66  4867.8 1669.13  4947.9 1667.53
  4977.9 1666.02  5044.9 1665.82  5045.4 1665.32  5050.4 1665.32  5050.9 1665.82
  5137.9  1667.2  5187.9 1668.56  5225.4 1669.99    5258 1670.15    5278 1670.79
    5308  1672.9    5328 1672.77    5378 1674.78    5428 1675.23  5437.4 1675.81
#Mann= 3 ,-1 , 0
  4626.1     .05       0  5044.9     .03       0  5050.9     .05       0
Bank Sta=5044.9,5050.9
XS Rating Curve= 0 ,0
Exp/Cntr=0.3,0.1

Type RM Length L Ch R = 1 ,31667   ,207,207,207
BEGIN DESCRIPTION:
Mapping XS db4b9baa
END DESCRIPTION:
XS GIS Cut Line= 2
      1594040.76      6948309.33      1594807.93      6947873.36
#Sta/Elev= 30
    4496 1675.68  4513.5 1674.53  4523.6 1672.21  4566.8 1671.26  4572.6  1671.6
  4588.5 1670.48  4610.1 1671.72    4626 1669.81  4631.7 1669.71  4638.9 1667.94
  4647.6 1666.89  4669.2 1665.85  4880.4 1661.75  4938.8 1661.84    4981 1661.17
  4981.5 1660.67  4986.5 1660.67    4987 1661.17    5007 1661.72  5029.6 1661.34
  5094.5 1662.76  5100.2 1663.38    5132 1663.35  5137.7    1664    5168 1663.93
  5202.6 1665.95    5256 1666.97  5283.3 1668.75  5336.7 1669.52  5378.4 1670.91
#Mann= 3 ,-1 , 0
    4496     .05       0    4981     .05       0    4987     .05       0
Bank Sta=4981,4987
XS Rating Curve= 0 ,0
Exp/Cntr=0.3,0.1

Type RM Length L Ch R = 1 ,31460   ,304,304,304
BEGIN DESCRIPTION:
Mapping XS 95a7ff44
END DESCRIPTION:
XS GIS Cut Line= 3
      1594163.61      6948523.55      1594736.06      6948111.71
      1594825.97      6947911.47
#Sta/Elev= 30
  4520.9 1672.32  4533.9 1672.38  4560.9 1671.14  4590.3 1670.98  4862.8 1661.27
  4883.7    1661  4898.4 1660.22  4941.5 1659.48  4945.7 1659.12  4946.2 1658.62
  4951.3 1658.62  4951.8 1659.12  4984.4 1659.47  4990.7 1659.21  5070.3 1660.37
    5085 1659.88  5105.9 1660.25  5120.6 1659.97  5206.5  1660.9  5241.2 1661.84
  5258.9 1663.45  5264.3 1663.21  5310.7 1664.18  5317.9 1664.83  5333.8 1665.31
  5339.8 1665.91    5357 1666.66  5385.7 1667.31    5432 1669.67  5445.6  1669.8
#Mann= 3 ,-1 , 0
  4520.9     .05       0  4945.7     .05       0  4951.8     .05       0
Bank Sta=4945.7,4951.8
XS Rating Curve= 0 ,0
Exp/Cntr=0.3,0.1

Type RM Length L Ch R = 1 ,31156   ,341,341,341
BEGIN DESCRIPTION:
Deadman 02 49.0
END DESCRIPTION:
XS GIS Cut Line= 3
        1594355.        6948838.        1594705.        6948488.
      1594954.99      6947738.04
#Sta/Elev= 30
  4505.5 1675.27  4590.4 1671.75  4731.8 1663.56  4816.6 1660.61  4844.9 1660.32
  4859.1 1659.37  4986.3 1655.86  5042.6 1656.53  5053.2 1656.01  5095.3  1655.9
  5102.8 1655.37  5103.3 1654.87  5108.5 1654.87    5109 1655.37  5137.5 1656.38
  5253.5 1657.73  5306.2 1659.04  5337.8 1660.57  5358.9 1660.74  5432.7 1663.81
  5464.3 1664.59  5527.5  1667.9  5548.6 1668.11  5590.8 1670.05  5601.3 1669.88
    5654 1672.82  5675.1 1672.97  5706.7 1674.79  5748.9 1675.32    5791 1677.63
#Mann= 3 ,-1 , 0
  4505.5     .05       0  5102.8     .05       0    5109     .05       0
Bank Sta=5102.8,5109
XS Rating Curve= 0 ,0
Exp/Cntr=0.3,0.1

Type RM Length L Ch R = 1 ,30815   ,252,252,252
BEGIN DESCRIPTION:
Mapping XS 7e86afff
END DESCRIPTION:
XS GIS Cut Line= 3
      1594591.63      6948806.14       1595010.7      6948593.22
      1595189.66      6948022.58
#Sta/Elev= 30
  4472.6 1664.92  4487.6  1663.8  4541.9 1662.45  4675.4 1657.16  4734.4 1655.97
  4824.1 1652.65  4903.6 1651.04  4936.3 1651.08  4948.1 1649.28  4968.8 1649.17
  4970.9 1647.14  4971.4 1646.64  4977.1 1647.14  4979.6 1648.37  5006.5 1650.05
  5011.7  1648.5  5038.9  1650.2  5044.1 1648.73  5052.9 1650.44  5063.4 1650.89
    5109 1651.33  5173.9 1653.73  5211.5 1653.71  5308.8 1656.43  5341.2 1658.38
  5388.3  1659.4    5471 1663.27  5508.6 1664.11    5535  1666.3  5540.7 1666.17
#Mann= 3 ,-1 , 0
  4472.6     .05       0  4970.9     .05       0  4977.1     .05       0
Bank Sta=4970.9,4977.1
XS Rating Curve= 0 ,0
Exp/Cntr=0.3,0.1

Type RM Length L Ch R = 1 ,30563   ,92,92,92
BEGIN DESCRIPTION:
Deadman 02 48.0
END DESCRIPTION:
XS GIS Cut Line= 3
      1595243.89      6949103.54      1595264.17      6948586.47
      1595240.51      6947944.37
#Sta/Elev= 30
  4483.7 1661.09  4539.3 1659.29  4599.3 1656.51    4637 1655.62    4642 1655.94
  4669.4 1654.35  4739.4 1652.14  4769.5 1650.71  4789.5 1650.74  4839.5 1649.38
  4879.5 1649.96  4899.7 1648.83  4976.5 1648.03    4977 1647.53  4982.3 1647.53
  4982.8 1648.03  5119.7 1650.39  5199.8 1651.24  5299.8 1653.94  5369.9 1656.37
  5385.4 1657.55  5390.4 1657.14  5429.9 1659.07    5480 1660.66    5530 1663.45
    5560 1665.98    5570 1665.63    5610 1667.46  5620.1 1668.41  5643.7 1668.84
#Mann= 3 ,-1 , 0
  4483.7     .05       0  4976.5     .03       0  4982.8     .05       0
Bank Sta=4976.5,4982.8
XS Rating Curve= 0 ,0
Exp/Cntr=0.3,0.1

Type RM Length L Ch R = 1 ,30471   ,429,429,429
BEGIN DESCRIPTION:
Mapping XS c86db497
END DESCRIPTION:
XS GIS Cut Line= 2
      1595362.18      6948971.75      1595348.66      6948153.86
#Sta/Elev= 30
  4610.8 1654.04  4714.6 1651.08  4724.6 1650.95  4741.1 1650.33  4746.1 1650.44
  4764.6 1649.87  4854.6 1648.04  4904.6 1646.76  4961.4 1645.99  4961.9 1645.49
  4967.2 1645.49  4967.7 1645.99  5004.6  1646.2  5024.6 1646.69  5094.6 1647.26
  5134.6 1647.22  5154.6 1647.66  5224.6 1649.76  5274.6 1651.62  5304.6 1652.53
  5324.6 1654.55  5334.6 1654.71  5343.6 1654.43  5348.6 1654.49  5354.7 1655.25
  5364.7 1655.72  5374.7 1656.61  5414.7 1658.46  5424.2 1659.08  5428.8 1659.08
#Mann= 3 ,-1 , 0
  4610.8     .05       0  4961.4     .03       0  4967.7     .05       0
Bank Sta=4961.4,4967.7
XS Rating Curve= 0 ,0
Exp/Cntr=0.3,0.1

Type RM Length L Ch R = 1 ,30042   ,404,404,404
BEGIN DESCRIPTION:
Mapping XS cf7890d7
END DESCRIPTION:
XS GIS Cut Line= 2
       1595723.8      6948910.88      1595737.32      6948187.71
#Sta/Elev= 30
    4653 1646.76  4695.9 1646.18  4735.9 1646.06  4755.9 1645.69  4775.9 1645.13
  4825.9 1644.66  4905.9  1643.2  4965.9 1642.59  4992.8 1641.56  4993.3 1641.06
  4998.6 1641.06  4999.1 1641.56  5005.9 1641.96  5015.9 1641.82  5025.9 1641.92
    5066 1642.65    5096 1643.43    5106 1643.85    5126 1644.31    5176 1646.41
    5196 1647.05    5236 1648.94    5246 1649.65    5286 1651.34    5296 1652.39
    5306 1652.86    5316 1653.59    5356  1655.8  5373.7 1656.92  5376.3 1656.92
#Mann= 3 ,-1 , 0
    4653     .05       0  4992.8     .05       0  4999.1     .05       0
Bank Sta=4992.8,4999.1
XS Rating Curve= 0 ,0
Exp/Cntr=0.3,0.1

Type RM Length L Ch R = 1 ,29638   ,255,255,255
BEGIN DESCRIPTION:
Mapping XS 4804a419
END DESCRIPTION:
XS GIS Cut Line= 2
      1596038.11      6948904.13      1596156.39      6948248.51
#Sta/Elev= 30
  4670.6 1642.36    4687 1642.08  4697.2  1642.2  4707.3 1641.99  4727.6 1642.08
  4788.6  1641.8  4793.8 1641.55  4859.7 1640.62  4869.9 1640.17  4930.9 1639.48
  4998.8 1638.34  4999.3 1637.84  5004.6 1637.84  5005.1 1638.34  5023.3 1639.01
  5076.9 1640.35  5103.6 1641.29  5130.4 1641.91  5135.5  1641.8    5184 1643.48
  5189.1 1643.36  5215.4 1644.38  5235.7 1644.84  5242.6 1645.24  5247.7 1645.14
  5286.5 1646.26  5306.8 1646.56    5317 1646.89  5334.5 1648.23  5336.8 1648.23
#Mann= 3 ,-1 , 0
  4670.6     .05       0  4998.8     .05       0  5005.1     .05       0
Bank Sta=4998.8,5005.1
XS Rating Curve= 0 ,0
Exp/Cntr=0.3,0.1

Type RM Length L Ch R = 1 ,29383   ,300,300,300
BEGIN DESCRIPTION:
Mapping XS 87066316
END DESCRIPTION:
XS GIS Cut Line= 2
      1596280.35      6948910.65      1596403.89       6948218.8
#Sta/Elev= 30
  4722.2 1639.59  4778.9 1639.18  4785.8 1639.39  4826.5 1639.41  4891.7 1639.09
  4897.6 1638.77  4938.2 1638.05  4958.5  1637.3  5009.5 1636.47  5016.3 1635.89
  5016.8 1635.39  5022.2 1635.39  5022.7 1635.89  5039.8 1636.89  5063.4 1637.22
  5100.7 1638.39  5122.3 1638.51    5171 1639.61  5176.1  1639.5    5230 1640.88
    5235 1640.71  5273.4 1641.78  5283.6 1641.85  5288.9 1642.19    5294 1642.09
  5334.4 1642.92  5347.8 1642.86    5375 1643.28  5401.6  1644.8    5425 1644.91
#Mann= 3 ,-1 , 0
  4722.2     .05       0  5016.3     .05       0  5022.7     .05       0
Bank Sta=5016.3,5022.7
XS Rating Curve= 0 ,0
Exp/Cntr=0.3,0.1

Type RM Length L Ch R = 1 ,29083   ,494,494,494
BEGIN DESCRIPTION:
Mapping XS 1ac94856
END DESCRIPTION:
XS GIS Cut Line= 2
      1596828.94      6949414.49      1596504.49       6948167.4
#Sta/Elev= 30
  4148.3 1646.04    4155 1647.11  4165.3  1647.6  4182.3 1644.73  4187.5 1645.46
  4196.3 1643.78  4206.7 1642.72  4222.8 1641.75    4228 1641.95  4289.3 1639.71
    4310 1638.07  4330.7 1637.99  4339.2 1637.06  4392.7 1636.02  4444.3 1636.02
  4516.7  1634.8  4541.9 1635.17  4565.1 1632.55  4565.6 1632.05    4571 1632.05
  4571.5 1632.55  4577.2 1636.05  4609.6 1635.34  4901.4 1635.18  4982.5 1633.81
  5012.6 1634.12    5271  1639.6  5331.7 1640.12  5353.6 1641.31  5436.9  1643.4
#Mann= 3 ,-1 , 0
  4148.3     .05       0  4565.1     .05       0  4571.5     .05       0
Bank Sta=4565.1,4571.5
XS Rating Curve= 0 ,0
Exp/Cntr=0.3,0.1

Type RM Length L Ch R = 1 ,28589   ,561,561,561
BEGIN DESCRIPTION:
Mapping XS 772ec94d
END DESCRIPTION:
XS GIS Cut Line= 2
      1597234.48      6949022.41      1596937.08      6948008.53
#Sta/Elev= 30
  4494.8 1637.32  4507.7 1637.27  4551.5  1635.4  4613.1 1634.18  4624.5 1633.24
  4666.1 1632.01  4707.8 1631.36  4720.5 1629.27    4721 1628.77  4726.4 1628.77
  4726.9 1629.27  4728.9 1629.92  4739.1 1630.46  4749.5    1630  4762.3 1631.28
  4989.2 1630.61  5045.1 1631.56  5197.6 1632.65    5281  1632.8  5301.8 1633.67
  5322.7 1633.33  5353.9 1633.79  5361.3 1633.33  5385.2 1633.82  5394.7 1633.45
  5399.9 1633.79  5510.5 1634.21  5531.1 1634.42  5538.7 1634.94  5551.4 1634.79
#Mann= 3 ,-1 , 0
  4494.8     .05       0  4720.5    .035       0  4726.9     .05       0
Bank Sta=4720.5,4726.9
XS Rating Curve= 0 ,0
Exp/Cntr=0.3,0.1

Type RM Length L Ch R = 1 ,28028   ,411,411,411
BEGIN DESCRIPTION:
Mapping XS 800fc63b
END DESCRIPTION:
XS GIS Cut Line= 2
      1597788.72      6948677.68      1597261.51      6947876.72
#Sta/Elev= 30
  4659.3 1636.07  4712.2 1635.32  4718.8 1634.44  4799.5 1631.93  4826.6 1631.86
  4850.5 1630.78  4877.8 1630.36  4898.9  1630.5    4908  1629.9  4944.1 1628.71
  4980.3 1628.74  4986.3 1628.38  4994.1 1626.21  4997.5 1625.81    4998 1625.31
  5004.6 1625.31  5005.1 1625.81  5016.4  1626.2  5043.5 1628.25  5101.9 1628.08
    5161 1628.51  5209.6 1629.32  5218.2 1628.69  5224.2  1629.1  5239.3 1628.88
  5245.5 1628.22  5269.4 1628.19  5413.1 1630.29  5456.2 1630.14  5618.2 1630.71
#Mann= 3 ,-1 , 0
  4659.3     .05       0  4997.5     .05       0  5005.1     .05       0
Bank Sta=4997.5,5005.1
XS Rating Curve= 0 ,0
Exp/Cntr=0.3,0.1

Type RM Length L Ch R = 1 ,27617   ,316,316,316
BEGIN DESCRIPTION:
Mapping XS 71541e72
END DESCRIPTION:
XS GIS Cut Line= 2
      1598055.72      6948512.07      1597697.51      6947687.52
#Sta/Elev= 30
  4601.3 1631.15  4660.3 1630.36  4736.1 1628.43  4770.5 1628.44  4788.5 1627.41
  4823.8 1626.84  4846.3 1626.87  4900.1 1625.95    4911 1626.28  4945.6 1626.23
  4954.6 1625.25  4963.6 1625.13    4969 1626.01  4998.2 1625.66  5009.1 1625.01
  5012.1 1622.62  5012.6 1622.12  5019.2 1622.12  5019.7 1622.62  5021.4 1623.54
    5031 1623.17  5039.4 1625.27  5044.8 1623.01  5052.8 1624.95  5062.8 1625.65
  5074.6 1625.34  5205.4 1625.79  5303.5 1627.28  5394.9 1627.61  5500.3 1627.39
#Mann= 3 ,-1 , 0
  4601.3     .05       0  5012.1     .05       0  5019.7     .05       0
Bank Sta=5012.1,5019.7
XS Rating Curve= 0 ,0
Exp/Cntr=0.3,0.1

Type RM Length L Ch R = 1 ,27301   ,397,397,397
BEGIN DESCRIPTION:
Mapping XS 6f44eaf5
END DESCRIPTION:
XS GIS Cut Line= 2
       1598269.4      6948474.12      1598079.98       6947543.5
#Sta/Elev= 30
  4605.8 1627.84  4714.1 1626.48  4785.5 1624.66  4807.2 1625.31  4836.6 1624.25
  4857.8 1624.51  4867.2 1623.66  4897.8 1623.97  4908.4 1624.75  4928.4 1624.64
  4938.6 1624.11  4948.7  1624.7  4999.3 1623.46  5004.4 1622.95  5006.2 1620.88
  5006.7 1620.38  5013.4 1620.38  5013.9 1620.88  5020.2 1622.12  5030.5  1622.8
  5040.7 1624.63  5061.1 1623.85  5091.7  1624.3  5112.1 1623.82  5156.2    1624
  5224.3 1623.04  5409.1 1624.93  5448.9 1624.57  5489.7 1624.86  5555.5  1625.8
#Mann= 3 ,-1 , 0
  4605.8     .05       0  5006.2     .05       0  5013.9     .05       0
Bank Sta=5006.2,5013.9
XS Rating Curve= 0 ,0
Exp/Cntr=0.3,0.1

Type RM Length L Ch R = 1 ,26904   ,89,89,89
BEGIN DESCRIPTION:
Mapping XS b6f15bfd
END DESCRIPTION:
XS GIS Cut Line= 4
      1598555.92      6948562.85      1598539.02      6948028.83
       1598542.4      6947829.43      1598528.84      6947267.51
#Sta/Elev= 30
  4525.4 1623.24  4830.4  1621.7  4860.4 1622.24  4930.5 1622.34  4970.5 1623.31
  5000.5 1621.02  5020.5 1624.96  5027.2 1625.34  5032.2 1624.14  5050.5  1621.7
  5080.5 1619.93  5100.5 1620.99  5110.5 1622.73  5121.4    1626  5140.5  1627.1
  5160.5 1621.92  5170.5 1621.54  5176.6 1618.84  5177.1 1618.34    5184 1618.34
  5184.5 1618.84  5190.5 1619.99  5230.5 1621.75  5250.5 1621.09  5270.6 1621.92
  5310.6 1621.39  5370.6  1622.2  5470.6 1622.13  5500.6 1621.62  5821.2 1623.72
#Mann= 3 ,-1 , 0
  4525.4     .05       0  5176.6     .03       0  5184.5     .05       0
Bank Sta=5176.6,5184.5
XS Rating Curve= 0 ,0
Exp/Cntr=0.3,0.1

Type RM Length L Ch R = 1 ,26815   ,424,424,424
BEGIN DESCRIPTION:
Mapping XS bdfac55e
END DESCRIPTION:
XS GIS Cut Line= 4
      1598657.31      6948471.54      1598630.27      6948106.56
      1598626.89      6947795.63      1598640.01      6947223.21
#Sta/Elev= 30
  4616.2 1622.53    4710 1621.93  4790.2 1621.92  4840.4 1621.31  4870.4 1621.97
  4890.5 1621.54  4970.7 1621.85  4990.7 1621.45  5000.7 1620.83  5040.7 1621.87
  5080.7 1622.26  5130.7 1621.53  5150.7  1620.5  5180.8 1620.34  5186.8 1619.86
  5187.3 1619.36  5194.2 1619.36  5194.7 1619.86  5280.8 1620.05  5340.8 1620.68
  5390.8 1620.46  5400.8 1620.05  5470.8 1620.57  5490.8 1620.25  5540.8 1620.32
  5660.9 1620.91  5670.9  1621.3  5720.9  1620.9  5770.9 1621.47  5865.7 1621.69
#Mann= 3 ,-1 , 0
  4616.2     .05       0  5186.8     .03       0  5194.7     .05       0
Bank Sta=5186.8,5194.7
XS Rating Curve= 0 ,0
Exp/Cntr=0.3,0.1

Type RM Length L Ch R = 1 ,26391   ,309,309,309
BEGIN DESCRIPTION:
Mapping XS 6ff5a1f0
END DESCRIPTION:
XS GIS Cut Line= 3
      1599032.45      6948566.18      1599018.93      6948008.55
      1598961.35      6946981.16
#Sta/Elev= 30
  4622.1 1623.93  4770.3 1620.72  4860.4 1620.39  4880.4 1619.83  4890.4 1620.44
  4940.4  1619.2  4970.4 1619.74  4990.4 1618.81  5110.4 1620.23  5135.6 1619.24
  5140.6 1619.96  5160.4 1617.97  5170.4 1618.06  5177.7    1620  5190.5 1620.62
  5200.5 1619.57  5250.6 1618.76  5280.6 1617.54  5380.8 1617.16  5470.9 1618.58
  5611.1 1617.54  5647.2 1616.75  5647.7 1616.25  5654.6 1616.25  5655.1 1616.75
  5771.4 1617.23  6011.8  1619.4  6071.8 1619.24  6121.9 1620.29  6208.9  1620.6
#Mann= 3 ,-1 , 0
  4622.1     .05       0  5647.2     .05       0  5655.1     .05       0
Bank Sta=5647.2,5655.1
XS Rating Curve= 0 ,0
Exp/Cntr=0.3,0.1

Type RM Length L Ch R = 1 ,26082   ,785,785,785
BEGIN DESCRIPTION:
Mapping XS 76fb0c02
END DESCRIPTION:
XS GIS Cut Line= 3
      1599302.82      6948488.45       1599289.3      6947728.04
      1599187.74      6947094.56
#Sta/Elev= 30
  4599.2 1625.17  4849.7 1618.68  4859.7 1619.16  4889.7  1618.3  4909.7 1618.47
  4929.7 1617.71  4979.7 1617.93  4989.7 1617.79  4999.7 1616.65  5009.7 1617.82
  5029.7  1618.5  5079.7 1618.44  5099.7 1618.74  5129.7 1617.51  5139.7 1616.57
  5179.7 1616.14  5239.8 1615.97  5289.8 1616.49  5317.6 1615.91  5322.6 1616.14
  5531.9 1616.23  5623.1 1615.55  5704.1 1615.43  5760.5 1614.88    5761 1614.38
  5768.8 1614.38  5769.3 1614.88  5845.9 1615.67  5866.2 1616.62  6001.3 1617.58
#Mann= 3 ,-1 , 0
  4599.2     .05       0  5760.5     .05       0  5769.3     .05       0
Bank Sta=5760.5,5769.3
XS Rating Curve= 0 ,0
Exp/Cntr=0.3,0.1

Type RM Length L Ch R = 1 ,25297   ,734,734,734
BEGIN DESCRIPTION:
Mapping XS 3bc6f327
END DESCRIPTION:
XS GIS Cut Line= 3
      1600215.33      6948231.61      1599607.82       6947821.4
       1599303.2      6947082.57
#Sta/Elev= 30
  4493.7 1626.95  4546.6 1626.03  4554.4 1626.24  4567.6 1625.17  4612.5 1624.73
  4699.2 1622.42  4771.4 1619.84  4807.3 1618.18  4813.4 1616.57  4834.4    1614
  4906.3  1614.5  4928.5 1613.71  4957.2 1614.24  4982.7 1613.22  4983.2 1612.72
  4991.2 1612.72  4991.7 1613.22  4993.2 1614.79  5023.1 1615.64  5029.2 1615.15
  5065.1 1614.73  5131.1 1615.17  5316.9 1614.77  5406.8 1614.97  5436.1 1615.86
  5585.1 1614.35  5750.4 1614.16  5880.9 1614.88  5928.7 1616.51  6025.9 1616.59
#Mann= 3 ,-1 , 0
  4493.7     .05       0  4982.7     .05       0  4991.7     .05       0
Bank Sta=4982.7,4991.7
XS Rating Curve= 0 ,0
Exp/Cntr=0.3,0.1

Type RM Length L Ch R = 1 ,24563   ,545,545,545
BEGIN DESCRIPTION:
Mapping XS 298414b9
END DESCRIPTION:
XS GIS Cut Line= 3
      1600627.67      6947728.05      1600262.63      6947592.86
        1599330.        6947063.
#Sta/Elev= 30
  4597.1 1622.59  4653.3 1621.05  4669.2 1621.55  4685.3 1619.95  4749.2 1618.13
  4770.6 1616.81  4780.2 1617.93  4791.9 1618.08  4919.9 1612.48  4951.8 1612.86
  4981.6 1609.87  4982.1 1609.37  4990.7 1609.87  5003.6 1610.71  5009.4 1609.88
  5018.1 1611.21    5031 1610.69  5062.7 1611.66  5121.7 1610.84  5143.5 1611.73
    5230 1611.23  5294.8 1612.35  5413.1 1612.49  5434.7 1613.75  5450.6 1612.55
  5466.4 1612.38  5574.6  1612.5    5736 1615.08  5800.9 1614.45    6059 1616.91
#Mann= 3 ,-1 , 0
  4597.1     .05       0  4981.6     .05       0  4990.7     .05       0
Bank Sta=4981.6,4990.7
XS Rating Curve= 0 ,0
Exp/Cntr=0.3,0.1

Type RM Length L Ch R = 1 ,24018   ,533,533,533
BEGIN DESCRIPTION:
Mapping XS 495d3da6
END DESCRIPTION:
XS GIS Cut Line= 2
      1600600.57      6947413.72      1599804.54      6947002.22
#Sta/Elev= 30
    4465 1616.99  4538.8 1614.85  4628.9 1613.68  4718.9  1611.7    4764 1611.34
  4831.3 1609.67  4853.5 1610.42    4942 1610.06  5008.5 1608.89  5022.9 1610.03
  5030.6 1609.84  5036.3 1608.68  5045.4  1609.8  5052.8  1609.7  5053.7 1608.23
  5054.2 1607.73  5062.5 1607.73    5063 1608.23  5080.5 1610.03  5090.4 1610.03
  5102.7 1611.51  5124.8 1611.73  5141.3 1612.47  5163.5 1612.25  5191.7 1612.86
  5252.1 1612.93  5274.2 1613.56  5281.8 1612.81  5304.3 1612.53  5361.1 1612.89
#Mann= 3 ,-1 , 0
    4465     .05       0  5053.7     .05       0    5063     .05       0
Bank Sta=5053.7,5063
XS Rating Curve= 0 ,0
Exp/Cntr=0.3,0.1

Type RM Length L Ch R = 1 ,23485   ,777,777,777
BEGIN DESCRIPTION:
Mapping XS fd83ad1f
END DESCRIPTION:
XS GIS Cut Line= 3
      1600708.78      6947349.55      1600336.98      6946994.66
      1599485.34      6946643.19
#Sta/Elev= 30
    4110 1617.09  4142.2 1616.85  4226.8 1614.03  4311.7 1612.84  4474.7 1608.99
  4540.4 1608.12  4540.9 1607.62  4549.2 1607.62  4549.7 1608.12  4580.6 1608.63
  4615.9 1608.29    4691 1609.63  4712.7 1608.55  4866.9 1609.31  4950.7 1608.38
  4997.3 1609.19  5004.8 1608.35  5015.6 1608.35  5037.2 1608.75  5074.5 1612.42
  5112.9 1611.86    5181 1611.85  5228.9 1612.52  5329.3 1612.69  5364.7 1613.65
  5412.6 1613.93  5448.3 1615.24  5489.8 1615.04  5524.5 1616.48  5545.3 1616.62
#Mann= 3 ,-1 , 0
    4110     .05       0  4540.4     .05       0  4549.7     .05       0
Bank Sta=4540.4,4549.7
XS Rating Curve= 0 ,0
Exp/Cntr=0.3,0.1

Type RM Length L Ch R = 1 ,22708   ,782,782,782
BEGIN DESCRIPTION:
Mapping XS 6a6bf8fa
END DESCRIPTION:
XS GIS Cut Line= 2
      1600911.54      6946933.84      1599777.63      6946242.02
#Sta/Elev= 30
  4560.4 1614.53  4678.3 1611.54  4809.9  1609.2  4883.5 1607.26  4999.6 1606.65
  5005.5  1607.1  5016.2 1606.24  5016.7 1605.74  5025.1 1605.74  5025.6 1606.24
  5026.8 1606.91  5042.3 1607.06  5173.9 1607.25    5232  1607.9  5282.6  1606.9
  5363.6 1607.28  5369.5 1606.46  5412.1 1607.66  5434.9 1607.29  5479.8 1607.86
  5485.6  1607.4  5528.6  1608.8  5580.5  1608.5  5638.6 1609.43  5659.9 1609.19
  5675.3 1610.33  5696.7 1610.85  5727.6 1612.64  5791.5 1612.54  5888.7 1614.07
#Mann= 3 ,-1 , 0
  4560.4     .05       0  5016.2     .05       0  5025.6     .05       0
Bank Sta=5016.2,5025.6
XS Rating Curve= 0 ,0
Exp/Cntr=0.3,0.1

Type RM Length L Ch R = 1 ,21926   ,898,898,898
BEGIN DESCRIPTION:
Mapping XS 91b51c6e
END DESCRIPTION:
XS GIS Cut Line= 2
      1601114.31      6946453.93        1600141.      6945710.43
#Sta/Elev= 30
  4478.8 1613.11  4540.4 1611.31  4603.8 1610.61  4617.4 1609.44    4690 1608.32
  4731.7 1606.61  4953.9 1605.27  4981.3 1603.83  4989.3 1604.91  5010.1 1603.37
  5024.6 1603.42  5039.2 1604.98  5074.5 1605.31  5095.3 1604.49  5104.5 1602.49
    5105 1601.99  5115.2 1602.49  5132.3 1604.73  5153.5 1605.36  5373.8  1605.9
  5452.7 1607.82  5481.8 1609.25  5502.6 1609.36    5567 1613.49  5573.3 1613.26
  5660.5 1617.96  5666.8 1617.59  5681.3 1618.93  5687.6  1618.2  5703.6 1618.88
#Mann= 3 ,-1 , 0
  4478.8     .05       0  5104.5     .05       0  5115.2     .05       0
Bank Sta=5104.5,5115.2
XS Rating Curve= 0 ,0
Exp/Cntr=0.3,0.1

Type RM Length L Ch R = 1 ,21028   ,421,421,421
BEGIN DESCRIPTION:
Mapping XS c5cb1baf
END DESCRIPTION:
XS GIS Cut Line= 3
      1601469.11      6945598.87      1601019.67      6945515.68
      1600201.75      6945397.39
#Sta/Elev= 30
  4558.2 1605.88  4647.1 1604.49  4694.6 1604.84  4705.1 1603.56  4868.9 1601.81
  4916.7 1601.61  4969.2 1602.44  4974.3 1600.63  4974.8 1600.13  4984.7 1600.13
  4985.2 1600.63  4989.5 1601.34  5015.1 1602.24  5050.3 1602.59  5240.4 1602.37
  5302.9 1601.68  5315.8 1600.84  5353.4    1602  5386.1 1601.89  5403.9 1602.82
  5515.1 1603.35  5555.5 1605.02  5596.9 1604.96  5636.3 1607.04  5667.2  1606.5
    5697 1608.39  5757.6 1609.16  5777.8 1610.09  5787.9  1611.8  5841.7 1611.96
#Mann= 3 ,-1 , 0
  4558.2     .05       0  4974.3     .05       0  4985.2     .05       0
Bank Sta=4974.3,4985.2
XS Rating Curve= 0 ,0
Exp/Cntr=0.3,0.1

Type RM Length L Ch R = 1 ,20607   ,461,461,461
BEGIN DESCRIPTION:
Mapping XS 4592e3fc
END DESCRIPTION:
XS GIS Cut Line= 3
       1601695.6      6945477.21       1601097.4      6945267.67
      1600128.75      6945119.17
#Sta/Elev= 30
  4505.9 1611.57  4515.2 1610.36  4577.3 1609.06  4582.6 1609.48  4707.8 1604.59
    4782 1602.99  4962.1 1601.62  4975.2 1600.85  4983.3 1599.59  4993.9 1599.31
  5000.9 1600.32  5015.1 1599.76  5037.2 1601.83  5057.5 1600.71    5094 1600.48
  5202.9 1601.47  5314.1  1600.3  5395.1 1601.28  5415.3 1600.71  5427.1 1598.54
  5427.6 1598.04    5438 1598.54  5465.9  1600.3    5648  1602.1  5850.3 1605.41
  6052.7 1609.78    6083 1609.84  6103.3 1610.59  6113.4 1612.22  6119.7 1611.57
#Mann= 3 ,-1 , 0
  4505.9     .05       0  5427.1     .05       0    5438     .05       0
Bank Sta=5427.1,5438
XS Rating Curve= 0 ,0
Exp/Cntr=0.3,0.1

Type RM Length L Ch R = 1 ,20146   ,311,311,311
BEGIN DESCRIPTION:
Deadman 02 32.0
END DESCRIPTION:
XS GIS Cut Line= 3
      1601955.01        6945438.      1601188.65      6944966.89
        1600355.        6944588.
#Sta/Elev= 30
  4091.5 1623.49  4094.4 1623.49  4099.2 1620.18  4120.5 1618.96  4135.9 1615.78
  4157.2  1617.7  4185.4 1617.47  4208.9 1615.41  4236.5 1615.72  4279.3 1613.19
  4367.9 1611.14  4549.3  1603.3  4643.2 1601.03  4701.9 1601.69  4767.9 1598.71
  4810.5 1600.19  4984.5 1599.61    4995 1597.23  4995.5 1596.73    5006 1597.23
  5023.6 1599.36    5039 1599.48  5203.8 1599.08  5242.2 1597.66  5265.3 1599.04
  5346.6 1599.92  5558.6 1600.04    5742 1605.31  5869.4 1612.18  5906.8 1613.12
#Mann= 3 ,-1 , 0
  4091.5     .05       0    4995     .05       0    5006     .05       0
Bank Sta=4995,5006
XS Rating Curve= 0 ,0
Exp/Cntr=0.3,0.1

Type RM Length L Ch R = 1 ,19835   ,236,236,236
BEGIN DESCRIPTION:
Mapping XS b142fc7e
END DESCRIPTION:
XS GIS Cut Line= 2
      1601865.25      6944854.17      1600411.82      6944487.37
#Sta/Elev= 30
  4318.3 1613.23  4323.4 1613.17  4339.2 1609.43  4349.5  1608.2  4364.5 1607.97
  4370.1 1606.68  4405.5  1605.9  4452.6 1603.13  4504.2 1601.21  4586.7 1600.28
  4610.8 1597.91  4638.3 1597.82  4651.9 1598.72  4934.1 1598.54  4980.4  1597.8
  4993.8 1595.04  4994.3 1594.54  5004.8 1595.04  5016.3 1597.47  5040.5 1598.31
  5215.8 1598.17  5246.8 1597.13    5288 1598.06  5339.6 1597.16  5370.5 1598.43
    5453 1599.25  5591.1 1602.51  5714.3    1607  5783.1 1611.19  5817.3 1611.83
#Mann= 3 ,-1 , 0
  4318.3     .05       0  4993.8     .05       0  5004.8     .05       0
Bank Sta=4993.8,5004.8
XS Rating Curve= 0 ,0
Exp/Cntr=0.3,0.1

Type RM Length L Ch R = 1 ,19599   ,518,518,518
BEGIN DESCRIPTION:
Mapping XS f5a90c2c
END DESCRIPTION:
XS GIS Cut Line= 2
      1601824.03      6944624.93      1600585.99      6944294.78
#Sta/Elev= 30
  4468.6 1606.04  4498.6  1604.3  4519.7 1604.36  4549.5 1600.79  4554.6 1598.91
  4560.7 1598.07  4589.6  1601.6  4594.7 1600.38  4602.1 1600.89  4612.5 1603.04
  4622.8 1603.93  4629.7 1603.05  4634.8  1603.6  4664.2 1597.84  4674.9 1597.21
  4865.1 1596.44  4974.7 1596.84  5015.2 1594.89  5036.8 1597.14    5161 1597.52
  5250.6 1596.53  5255.8 1594.79    5259  1594.6  5259.5  1594.1    5270  1594.6
  5305.9 1598.53  5347.3 1596.75    5521 1598.86  5730.2 1605.46  5749.9 1605.47
#Mann= 3 ,-1 , 0
  4468.6     .05       0    5259     .03       0    5270     .05       0
Bank Sta=5259,5270
XS Rating Curve= 0 ,0
Exp/Cntr=0.3,0.1

Type RM Length L Ch R = 1 ,19081   ,385,385,385
BEGIN DESCRIPTION:
Mapping XS 8a35169a
END DESCRIPTION:
XS GIS Cut Line= 3
      1602007.37       6944290.2      1601428.52      6944153.48
      1600518.14      6944192.68
#Sta/Elev= 30
  4637.9 1609.38  4641.7 1609.38  4667.6 1605.65  4752.2 1602.05  4757.4 1602.61
  4773.9 1602.09  4799.7 1600.52  4926.6 1597.11    5000  1594.2  5058.6 1594.36
  5086.8  1593.2  5087.3  1592.7  5097.5  1592.7    5098  1593.2  5164.4 1594.86
    5226 1594.87  5256.2 1595.83  5306.3 1594.88  5326.3 1596.29  5346.3 1596.42
  5356.3 1595.44  5376.3 1597.99  5396.3 1594.16  5416.4 1593.51  5446.4 1595.49
  5596.5 1594.69  5626.6 1595.51    5689 1595.75  5915.3  1600.7  6143.9 1607.44
#Mann= 3 ,-1 , 0
  4637.9     .05       0  5086.8     .05       0    5098     .05       0
Bank Sta=5086.8,5098
XS Rating Curve= 0 ,0
Exp/Cntr=0.3,0.1

Type RM Length L Ch R = 1 ,18696   ,427,427,427
BEGIN DESCRIPTION:
Mapping XS f0c6221c
END DESCRIPTION:
XS GIS Cut Line= 3
      1602264.17      6943946.34      1601617.66      6943836.29
      1600471.41      6943795.03
#Sta/Elev= 30
  4336.3 1608.02  4353.4 1608.32  4406.5 1606.88  4426.8 1604.97    4447 1604.97
  4487.6 1602.95  4568.8 1601.55  4609.3 1598.16  4654.6 1597.46  4660.1 1596.77
  4731.1 1594.81  4791.9 1593.45  4933.9 1594.09  4955.7  1593.6  4974.5 1591.81
  4995.9 1593.06  5004.8 1592.15  5029.2 1591.55  5029.7 1591.05  5040.4 1591.55
  5054.8 1593.26  5174.9 1593.41  5224.9 1591.83    5275 1594.48    5315 1593.69
    5345 1594.49  5485.1 1594.19  5595.2 1595.57  5735.3  1596.2  6139.1 1602.36
#Mann= 3 ,-1 , 0
  4336.3     .05       0  5029.2     .05       0  5040.4     .05       0
Bank Sta=5029.2,5040.4
XS Rating Curve= 0 ,0
Exp/Cntr=0.3,0.1

Type RM Length L Ch R = 1 ,18269   ,467,467,467
BEGIN DESCRIPTION:
Mapping XS 1cee4d2d
END DESCRIPTION:
XS GIS Cut Line= 3
      1602365.04      6943703.34      1601718.53      6943437.39
      1600604.38      6943565.77
#Sta/Elev= 30
    4281 1604.76  4332.1 1603.93  4337.5 1602.93    4356 1602.64  4385.4  1600.6
  4414.8 1601.42  4432.4 1599.27    4516 1595.79  4699.9 1593.07  4782.6 1592.69
  4800.1 1593.49    4812 1592.68  4961.1 1591.93  4993.7 1590.85    5008 1589.49
  5008.5 1588.99  5019.6 1589.49    5034 1591.24  5064.2 1592.08  5104.4 1591.28
  5201.9 1591.12  5235.3 1592.54  5305.7 1593.23  5335.9 1593.34    5346 1592.52
  5374.8 1594.13  5379.9 1593.45  5468.8  1594.6    5799 1596.01  6101.6 1598.84
#Mann= 3 ,-1 , 0
    4281     .05       0    5008     .05       0  5019.6     .05       0
Bank Sta=5008,5019.6
XS Rating Curve= 0 ,0
Exp/Cntr=0.3,0.1
