--- Deadman 17.prj (project) ---

Proj Title=Deadman 17 Base Level Engineering
Current Plan=p01
Default Exp/Contr=0.3,0.1
English Units
Geom File=g01
Flow File=f01
Plan File=p01
BEGIN DESCRIPTION:
Deadman 17
END DESCRIPTION:

--- Deadman 17.p01 (plan) ---

Plan Title=Multiple Run
Short Identifier=Multiple
Geom File=g01
Flow File=f01
Subcritical Flow
K Sum by GR= 0
Std Step Tol= 0.01
Critical Tol= 0.01
Num of Std Step Trials= 20
Max Error Tol= 0.3
Flow Tol Ratio= 0.001
Split Flow NTrial= 30
Split Flow Tol= 0.02
Split Flow Ratio= 0.02
Log Output Level= 0
Friction Slope Method= 1
Unsteady Friction Slope Method= 2
Unsteady Bridges Friction Slope Method= 1
Parabolic Critical Depth
Global Vel Dist=  1 , 1 , 1
Global Log Level= 0
CheckData=True
Encroach Param= -1, 0, 0, 0
BEGIN DESCRIPTION:
Multiple Run
END DESCRIPTION:

--- Deadman 17.f01 (steady flow) ---

Flow Title=Multiple
Number of Profiles=7
Profile Names=10-year,25-year,50-year,1pct_min,100-year,1pct_plu,500-year
River Rch & RM= Deadman 17,Reach-1,92876
     117     148     171      98     196     391     260
River Rch & RM= Deadman 17,Reach-1,88445
     292     395     477     286     571    1139     829
River Rch & RM= Deadman 17,Reach-1,85045
     311     420     507     303     605    1207     874
River Rch & RM= Deadman 17,Reach-1,79267
     408     557     676     406     811    1618    1184
River Rch & RM= Deadman 17,Reach-1,74077
     434     593     721     434     867    1729    1270
River Rch & RM= Deadman 17,Reach-1,65695
     537     741     905     548    1093    2181    1616
River Rch & RM= Deadman 17,Reach-1,61073
     596     827    1016     618    1233    2460    1841
River Rch & RM= Deadman 17,Reach-1,58439
     881    1245    1549     953    1902    3794    2907
River Rch & RM= Deadman 17,Reach-1,46106
     883    1246    1548     951    1898    3786    2893
River Rch & RM= Deadman 17,Reach-1,42358
     856    1202    1490     913    1821    3633    2760
River Rch & RM= Deadman 17,Reach-1,39073
     929    1308    1623     996    1987    3964    3018
River Rch & RM= Deadman 17,Reach-1,36940
     882    1234    1523     930    1855    3702    2791
River Rch & RM= Deadman 17,Reach-1,19946
    1044    1478    1841    1133    2261    4511    3459
River Rch & RM= Deadman 17,Reach-1,14108
    1077    1527    1903    1173    2340    4670    3589
River Rch & RM= Deadman 17,Reach-1,12802
    1213    1733    2171    1345    2684    5356    4159
River Rch & RM= Deadman 17,Reach-1,7370
    1245    1781    2234    1385    2764    5515    4291
River Rch & RM= Deadman 17,Reach-1,268
    1237    1767    2215    1372    2738    5463    4242
Boundary for River Rch & Prof#=Deadman 17,Reach-1,1
Up Type=0
Dn Type=3
Dn Slope=0.005
Boundary for River Rch & Prof#=Deadman 17,Reach-1,2
Up Type=0
Dn Type=3
Dn Slope=0.005
Boundary for River Rch & Prof#=Deadman 17,Reach-1,3
Up Type=0
Dn Type=3
Dn Slope=0.005
Boundary for River Rch & Prof#=Deadman 17,Reach-1,4
Up Type=0
Dn Type=3
Dn Slope=0.005
Boundary for River Rch & Prof#=Deadman 17,Reach-1,5
Up Type=0
Dn Type=3
Dn Slope=0.005
Boundary for River Rch & Prof#=Deadman 17,Reach-1,6
Up Type=0
Dn Type=3
Dn Slope=0.005
Boundary for River Rch & Prof#=Deadman 17,Reach-1,7
Up Type=0
Dn Type=3
Dn Slope=0.005

--- Deadman 17.g01 (geometry) ---

Geom Title=Existing Conditions

River Reach=Deadman 17,Reach-1
Reach XY= 30
      1577955.00      6941938.00      1574717.92      6940901.50
      1572597.15      6936381.81      1571088.32      6935921.36
      1570704.49      6934567.79      1573111.21      6934230.24
      1575248.06      6931446.83      1576394.52      6931787.07
      1579791.78      6930201.67      1579597.49      6928134.83
      1578115.95      6927398.38      1577612.77      6925834.59
      1579096.03      6923731.30      1578306.56      6923031.91
      1578638.82      6922171.30      1577651.68      6921746.04
      1576557.55      6923183.01      1574977.36      6923261.70
      1574041.60      6921024.67      1572155.00      6919788.00
      1569856.50      6912843.82      1570562.76      6910331.83
      1572535.77      6908808.57      1574091.64      6905401.41
      1577865.32      6905377.17      1578252.03      6904093.52
      1579753.78      6903934.63      1582487.83      6901154.11
      1583564.70      6901027.23      1584305.00      6899288.00

Type RM Length L Ch R = 1,92876,643,643,643
BEGIN DESCRIPTION:
Mapping XS c2063c78
END DESCRIPTION:
XS GIS Cut Line= 3
      1578284.03      6940865.15      1577837.92      6941921.24
      1577419.69      6943012.28
#Sta/Elev= 30
  3854.2 1732.19  3892.8 1732.72  4022.2 1728.44  4259.0 1725.33  4375.7 1721.34
  4399.4 1721.05  4404.9 1722.62  4428.6 1720.82  4434.0 1722.04  4476.0 1720.74
  4481.4 1721.98  4541.2 1717.87  4639.9 1715.99  4996.0 1715.18  4996.5 1714.18
  5004.0 1715.18  5147.1 1715.30  5187.5 1718.22  5254.2 1718.44  5618.3 1727.91
  5736.1 1728.07  5745.3 1728.45  5768.3 1733.49  5789.7 1734.56  5860.1 1728.81
  5865.5 1727.17  5890.1 1726.55  6046.7 1726.73  6109.0 1729.15  6169.1 1727.72
#Mann=3,-1,0
  3854.2    0.05       0  4996.0    0.05       0  5004.0    0.05       0
Bank Sta=4996,5004
Exp/Cntr=0.3,0.1

Type RM Length L Ch R = 1,92233,999,999,999
BEGIN DESCRIPTION:
Mapping XS b3a56b8c
END DESCRIPTION:
XS GIS Cut Line= 2
      1577573.91      6940701.32      1576918.42      6942822.55
#Sta/Elev= 30
  3910.8 1732.68  4091.9 1728.29  4181.2 1727.95  4304.8 1723.69  4388.8 1724.63
  4504.5 1719.93  4531.9 1723.59  4537.1 1722.04  4597.2 1719.21  4640.3 1723.37
  4700.3 1716.94  4996.0 1715.18  4996.5 1714.18  5003.5 1714.18  5004.0 1715.18
  5112.9 1715.55  5205.2 1717.69  5236.6 1719.47  5288.9 1725.77  5308.7 1724.56
  5313.9 1726.18  5330.8 1721.90  5341.2 1720.94  5487.8 1725.51  5780.8 1727.73
  5812.2 1732.10  5833.2 1732.53  5864.6 1730.09  5906.4 1729.41  6131.0 1730.93
#Mann=5,-1,0
  3910.8    0.05       0  4181.2    0.12       0  4304.8    0.05       0
  4996.0    0.05       0  5004.0    0.05       0
Bank Sta=4996,5004
Exp/Cntr=0.3,0.1

Type RM Length L Ch R = 1,91234,338,338,338
BEGIN DESCRIPTION:
Mapping XS f2c79a71
END DESCRIPTION:
XS GIS Cut Line= 3
      1576693.98      6940775.63      1576317.55      6941501.20
      1576293.24      6941910.97
#Sta/Elev= 30
  4146.0 1725.50  4198.7 1725.68  4205.0 1726.36  4281.6 1725.99  4317.7 1726.53
  4392.2 1725.20  4420.0 1726.37  4436.4 1725.83  4486.6 1726.54  4541.4 1725.86
  4547.1 1726.53  4666.9 1725.31  4679.8 1725.97  4696.3 1725.62  4724.0 1726.54
  4790.8 1726.96  4829.0 1726.81  4858.4 1725.53  4903.5 1724.75  4970.2 1725.41
  4996.0 1724.62  4996.5 1723.62  5003.5 1723.62  5004.0 1724.62  5010.3 1725.34
  5030.3 1725.58  5060.4 1725.19  5190.6 1726.96  5300.8 1727.32  5373.9 1729.74
#Mann=3,-1,0
  4146.0    0.05       0  4996.0    0.05       0  5004.0    0.05       0
Bank Sta=4996,5004
Exp/Cntr=0.3,0.1

Type RM Length L Ch R = 1,90896,304,304,304
BEGIN DESCRIPTION:
Mapping XS 5e9df54f
END DESCRIPTION:
XS GIS Cut Line= 3
      1576580.01      6940562.99      1576022.41      6941410.92
      1575775.99      6942063.39
#Sta/Elev= 30
  3903.9 1725.54  4157.0 1725.59  4193.1 1724.90  4214.2 1725.58  4343.7 1724.80
  4467.3 1725.83  4509.4 1725.06  4684.2 1726.95  4879.3 1725.50  4969.1 1726.83
  4990.5 1728.17  4996.0 1724.80  4996.5 1723.80  5003.5 1723.80  5004.0 1724.80
  5008.5 1728.13  5033.2 1727.88  5063.5 1728.84  5068.9 1728.04  5086.7 1728.85
  5099.0 1728.00  5123.9 1728.43  5129.4 1729.23  5233.9 1729.63  5324.5 1728.34
  5404.4 1729.07  5503.5 1726.50  5535.6 1727.44  5549.9 1726.70  5616.2 1727.38
#Mann=3,-1,0
  3903.9    0.05       0  4996.0    0.05       0  5004.0    0.05       0
Bank Sta=4996,5004
Exp/Cntr=0.3,0.1

Type RM Length L Ch R = 1,90592,198,198,198
BEGIN DESCRIPTION:
Mapping XS f53bca3d
END DESCRIPTION:
XS GIS Cut Line= 2
      1576080.00      6940112.98      1575567.54      6941931.77
#Sta/Elev= 30
  3661.9 1725.69  3719.1 1726.49  3769.2 1725.14  3823.0 1728.68  3895.7 1725.73
  4067.3 1724.75  4124.2 1725.51  4174.6 1723.47  4269.7 1724.05  4394.3 1722.82
  4477.9 1724.62  4506.7 1722.74  4810.1 1721.91  4917.3 1722.56  4945.0 1724.39
  4956.5 1722.88  4990.5 1723.96  4996.0 1721.91  4996.5 1720.91  5003.5 1720.91
  5004.0 1721.91  5007.3 1724.12  5163.2 1724.76  5194.3 1726.90  5210.3 1725.31
  5288.7 1723.74  5402.1 1726.06  5474.9 1725.28  5508.4 1726.69  5551.5 1726.49
#Mann=3,-1,0
  3661.9    0.05       0  4996.0    0.05       0  5004.0    0.05       0
Bank Sta=4996,5004
Exp/Cntr=0.3,0.1

Type RM Length L Ch R = 1,90394,358,358,358
BEGIN DESCRIPTION:
Mapping XS 76d17965
END DESCRIPTION:
XS GIS Cut Line= 2
      1575879.99      6939963.05      1575387.00      6941938.67
#Sta/Elev= 30
  3556.4 1726.96  3613.0 1725.93  3654.3 1723.09  3721.4 1724.49  4056.7 1722.80
  4159.3 1725.91  4180.5 1725.73  4200.5 1723.45  4304.3 1722.00  4375.7 1723.01
  4602.5 1719.01  4629.2 1720.60  4684.9 1719.58  4711.8 1721.37  4716.9 1720.44
  4736.5 1721.41  4799.5 1719.20  4994.1 1720.83  4996.0 1719.01  4996.5 1718.01
  5003.5 1718.01  5004.0 1719.01  5005.8 1721.35  5076.6 1722.29  5406.4 1723.99
  5427.0 1722.93  5488.8 1724.02  5550.7 1730.34  5578.3 1724.47  5592.6 1724.07
#Mann=3,-1,0
  3556.4    0.05       0  4996.0    0.03       0  5004.0    0.05       0
Bank Sta=4996,5004
Exp/Cntr=0.3,0.1

Type RM Length L Ch R = 1,90036,1591,1591,1591
BEGIN DESCRIPTION:
Mapping XS a5af79b1
END DESCRIPTION:
XS GIS Cut Line= 3
      1575661.29      6939900.53      1575196.02      6941282.45
      1575084.90      6941827.60
#Sta/Elev= 30
  3546.3 1723.86  3596.4 1725.59  3612.6 1723.63  3670.2 1720.67  3764.8 1721.53
  3896.1 1719.69  4102.9 1719.00  4166.2 1722.56  4218.9 1719.51  4400.0 1716.84
  4725.4 1717.91  4804.2 1716.41  4873.1 1717.65  4893.4 1716.63  4993.2 1716.67
  4996.0 1715.73  4996.5 1714.73  5003.5 1714.73  5004.0 1715.73  5035.1 1716.85
  5153.0 1715.73  5275.5 1716.33  5397.9 1720.33  5439.5 1720.37  5459.2 1722.21
  5490.0 1721.66  5510.2 1723.57  5520.4 1726.60  5540.8 1729.49  5560.8 1727.24
#Mann=3,-1,0
  3546.3    0.05       0  4996.0    0.05       0  5004.0    0.05       0
Bank Sta=4996,5004
Exp/Cntr=0.3,0.1

Type RM Length L Ch R = 1,88445,157,157,157
BEGIN DESCRIPTION:
Mapping XS 47a7d085
END DESCRIPTION:
XS GIS Cut Line= 4
      1575380.01      6939012.99      1574962.57      6939288.03
      1574727.26      6940325.37      1574455.65      6941643.68
#Sta/Elev= 30
  3699.0 1726.40  3930.9 1723.01  3973.0 1724.93  4160.1 1724.70  4280.9 1721.28
  4496.2 1721.80  4557.8 1718.83  4658.9 1718.19  4701.3 1718.57  4721.8 1720.95
  4762.8 1717.76  4841.6 1717.00  4884.7 1717.00  4896.1 1720.16  4932.9 1716.75
  4957.7 1717.84  4976.0 1712.25  4995.4 1711.60  4995.9 1710.60  5004.6 1711.60
  5029.4 1716.32  5193.5 1716.71  5255.2 1720.97  5294.7 1720.52  5316.3 1716.88
  5336.8 1716.39  6089.3 1716.64  6290.5 1722.31  6521.1 1724.39  6608.6 1727.86
#Mann=3,-1,0
  3699.0    0.05       0  4995.4    0.03       0  5004.6    0.05       0
Bank Sta=4995.4,5004.6
Exp/Cntr=0.3,0.1

Type RM Length L Ch R = 1,88288,121,121,121
BEGIN DESCRIPTION:
Mapping XS d1f1ff35
END DESCRIPTION:
XS GIS Cut Line= 3
      1575085.23      6939065.98      1574866.46      6939102.44
      1574303.05      6941611.26
#Sta/Elev= 30
  3901.7 1724.40  3972.9 1722.97  4121.7 1724.01  4487.9 1720.31  4549.4 1722.12
  4621.1 1720.43  4662.1 1721.50  4805.6 1720.05  4877.4 1721.36  4949.1 1719.05
  4990.1 1719.06  4995.4 1712.36  4995.9 1711.36  5004.1 1711.36  5004.6 1712.36
  5017.9 1718.18  5082.4 1717.60  5256.6 1719.85  5318.1 1719.13  5336.5 1720.43
  5379.6 1719.06  5410.3 1712.99  5420.6 1712.36  5492.3 1717.11  5594.8 1717.63
  5625.6 1719.09  5795.3 1718.01  6291.7 1720.33  6466.0 1723.57  6694.8 1725.62
#Mann=3,-1,0
  3901.7    0.05       0  4995.4    0.03       0  5004.6    0.05       0
Bank Sta=4995.4,5004.6
Exp/Cntr=0.3,0.1

Type RM Length L Ch R = 1,88167,240,240,240
BEGIN DESCRIPTION:
Mapping XS 0ac25ae8
END DESCRIPTION:
XS GIS Cut Line= 5
      1575064.43      6939062.17      1574855.71      6939092.87
      1574622.50      6939829.35      1573978.07      6940670.16
      1573339.87      6940860.40
#Sta/Elev= 30
  3962.4 1723.25  4101.9 1722.65  4173.4 1724.31  4472.4 1720.18  4758.2 1721.46
  4829.1 1719.33  4947.9 1721.41  4985.6 1720.21  4995.4 1718.72  4995.9 1717.72
  5004.1 1717.72  5004.6 1718.72  5007.2 1719.91  5085.3 1718.72  5263.9 1721.16
  5421.7 1720.42  5463.3 1722.49  5506.9 1720.47  5756.2 1722.35  5799.7 1724.03
  5970.1 1723.39  6185.4 1729.08  6300.6 1727.63  6328.5 1728.87  6471.5 1729.29
  6551.1 1731.49  6634.5 1730.95  6642.5 1733.43  6647.7 1732.49  6671.2 1736.93
#Mann=3,-1,0
  3962.4    0.05       0  4995.4    0.03       0  5004.6    0.05       0
Bank Sta=4995.4,5004.6
Exp/Cntr=0.3,0.1

Type RM Length L Ch R = 1,87927,308,308,308
BEGIN DESCRIPTION:
Mapping XS 1e41fddf
END DESCRIPTION:
XS GIS Cut Line= 5
      1575202.43      6938683.55      1574859.83      6939072.61
      1574833.31      6939082.55      1574564.87      6939622.76
      1573461.26      6940196.11
#Sta/Elev= 30
  3756.5 1722.20  3850.0 1722.58  3913.6 1721.30  4034.1 1722.38  4097.6 1721.96
  4197.2 1724.59  4290.7 1724.70  4352.0 1722.66  4492.0 1722.42  4598.4 1720.78
  4732.8 1720.49  4789.5 1721.37  4995.4 1719.89  4995.9 1718.89  5004.1 1718.89
  5004.6 1719.89  5086.6 1721.37  5147.1 1720.68  5289.4 1722.33  5312.0 1721.10
  5384.7 1722.50  5423.3 1721.52  5628.0 1725.50  5672.6 1724.21  5821.4 1724.62
  5964.9 1726.97  6009.1 1726.72  6067.0 1729.57  6103.2 1730.25  6150.1 1729.13
#Mann=3,-1,0
  3756.5    0.05       0  4995.4    0.05       0  5004.6    0.05       0
Bank Sta=4995.4,5004.6
Exp/Cntr=0.3,0.1

Type RM Length L Ch R = 1,87619,203,203,203
BEGIN DESCRIPTION:
Mapping XS fdd49578
END DESCRIPTION:
XS GIS Cut Line= 5
      1575182.42      6938608.47      1574846.57      6939039.47
      1574690.80      6939208.49      1574293.10      6939433.86
      1573391.69      6939881.25
#Sta/Elev= 30
  3734.9 1722.34  3768.7 1722.85  3804.0 1721.77  3824.8 1722.66  3932.4 1720.98
  3988.5 1722.05  4160.4 1722.67  4203.4 1724.21  4245.5 1723.26  4274.4 1724.48
  4516.2 1721.80  4677.8 1723.66  4736.2 1721.31  4758.6 1721.85  4807.6 1720.30
  4920.1 1719.43  4985.9 1720.19  4995.4 1719.43  4995.9 1718.43  5004.1 1718.43
  5004.6 1719.43  5254.8 1721.45  5277.2 1720.59  5350.0 1722.04  5568.5 1723.79
  5602.5 1725.06  5753.4 1724.85  5859.3 1726.31  5910.3 1728.23  5974.6 1727.90
#Mann=3,-1,0
  3734.9    0.05       0  4995.4    0.03       0  5004.6    0.05       0
Bank Sta=4995.4,5004.6
Exp/Cntr=0.3,0.1

Type RM Length L Ch R = 1,87416,420,420,420
BEGIN DESCRIPTION:
Mapping XS 98a76640
END DESCRIPTION:
XS GIS Cut Line= 4
      1575042.27      6938458.32      1574544.98      6939042.78
      1574405.79      6939162.09      1573219.62      6939755.18
#Sta/Elev= 30
  3731.4 1722.54  4041.5 1721.02  4119.9 1722.03  4162.3 1723.30  4200.2 1722.29
  4346.8 1723.77  4371.1 1723.01  4431.4 1724.66  4513.5 1723.08  4642.1 1723.18
  4765.1 1721.29  4832.8 1720.50  4989.6 1720.47  4995.4 1720.16  4995.9 1719.16
  5004.1 1719.16  5004.6 1720.16  5040.4 1720.55  5214.2 1721.02  5248.0 1720.54
  5438.8 1722.23  5455.6 1722.60  5551.1 1723.63  5647.9 1724.62  5709.4 1722.95
  5759.5 1724.84  5789.9 1725.96  5826.8 1725.22  5843.5 1726.24  6008.3 1726.67
#Mann=18,-1,0
  3731.4    0.12       0  4119.9    0.05       0  4200.2    0.12       0
  4371.1    0.05       0  4513.5    0.12       0  4642.1    0.05       0
  4765.1    0.12       0  4832.8    0.05       0  4989.6    0.12       0
  4995.4    0.07       0  5004.6    0.12       0  5040.4    0.05       0
  5214.2    0.12       0  5248.0    0.05       0  5438.8    0.12       0
  5455.6    0.05       0  5551.1    0.12       0  5759.5    0.05       0
Bank Sta=4995.4,5004.6
Exp/Cntr=0.3,0.1

Type RM Length L Ch R = 1,86996,620,620,620
BEGIN DESCRIPTION:
Mapping XS 46c74852
END DESCRIPTION:
XS GIS Cut Line= 2
      1574726.96      6938263.10      1573290.10      6939473.14
#Sta/Elev= 30
  3902.3 1725.16  3984.8 1725.38  4091.4 1723.39  4191.5 1727.21  4261.8 1725.60
  4467.3 1723.41  4573.9 1724.82  4638.7 1724.17  4715.7 1724.35  4766.3 1722.13
  4872.3 1722.83  4995.4 1721.41  4995.9 1720.41  5004.1 1720.41  5004.6 1721.41
  5042.3 1722.08  5099.3 1721.45  5148.7 1723.14  5210.9 1721.71  5234.5 1722.10
  5284.0 1724.94  5362.0 1724.47  5404.9 1726.12  5489.5 1723.21  5553.2 1724.27
  5596.1 1724.30  5603.9 1723.49  5631.2 1724.41  5752.2 1723.54  5780.8 1724.27
#Mann=5,-1,0
  3902.3    0.12       0  4638.7    0.05       0  4995.4    0.05       0
  5004.6    0.05       0  5210.9    0.12       0
Bank Sta=4995.4,5004.6
Exp/Cntr=0.3,0.1

Type RM Length L Ch R = 1,86376,550,550,550
BEGIN DESCRIPTION:
Mapping XS e0bfebfe
END DESCRIPTION:
XS GIS Cut Line= 3
      1574175.15      6938320.66      1573432.13      6938772.03
      1572825.81      6939264.02
#Sta/Elev= 30
  4134.0 1724.23  4424.1 1722.57  4583.1 1724.21  4619.9 1723.46  4672.2 1724.94
  4766.0 1721.67  4824.5 1722.50  4852.5 1720.80  4995.4 1720.78  4995.9 1719.78
  5004.1 1719.78  5004.6 1720.78  5019.9 1722.48  5119.0 1721.90  5226.1 1723.04
  5296.5 1721.92  5411.4 1723.50  5432.3 1724.88  5461.0 1723.68  5502.6 1725.72
  5531.4 1724.22  5609.7 1724.21  5619.6 1726.68  5624.1 1726.83  5630.7 1729.75
  5638.4 1730.83  5652.8 1728.64  5659.3 1725.62  5673.6 1723.70  5784.2 1724.54
#Mann=4,-1,0
  4134.0    0.05       0  4995.4    0.05       0  5004.6    0.05       0
  5619.6    0.12       0
Bank Sta=4995.4,5004.6
Exp/Cntr=0.3,0.1

Type RM Length L Ch R = 1,85826,781,781,781
BEGIN DESCRIPTION:
Mapping XS 391580c2
END DESCRIPTION:
XS GIS Cut Line= 3
      1574196.41      6937937.77      1573380.61      6938233.06
      1572665.30      6938523.18
#Sta/Elev= 30
  4071.0 1726.14  4103.9 1725.92  4210.7 1723.62  4253.3 1724.60  4321.9 1723.46
  4464.5 1723.93  4519.2 1722.44  4593.6 1723.06  4617.7 1722.10  4648.4 1722.60
  4735.0 1721.04  4790.9 1721.64  4995.4 1719.95  4995.9 1718.95  5004.1 1718.95
  5004.6 1719.95  5016.5 1720.82  5060.0 1720.27  5166.4 1720.74  5505.8 1722.34
  5522.9 1721.32  5559.7 1722.28  5606.0 1720.45  5630.0 1720.43  5667.7 1722.87
  5678.2 1722.77  5683.6 1723.98  5700.0 1724.10  5707.7 1723.88  5710.5 1721.69
#Mann=6,-1,0
  4071.0    0.12       0  4103.9    0.05       0  4995.4    0.05       0
  5004.6    0.05       0  5060.0    0.12       0  5166.4    0.05       0
Bank Sta=4995.4,5004.6
Exp/Cntr=0.3,0.1

Type RM Length L Ch R = 1,85045,978,978,978
BEGIN DESCRIPTION:
Mapping XS 95468e67
END DESCRIPTION:
XS GIS Cut Line= 3
      1573575.80      6937327.14      1572709.92      6937932.75
      1572164.47      6938413.15
#Sta/Elev= 30
  3971.7 1723.51  4058.1 1721.33  4141.3 1721.76  4199.8 1720.84  4368.8 1720.09
  4426.6 1720.48  4525.4 1722.11  4575.9 1720.32  4603.1 1720.89  4647.4 1722.11
  4712.9 1719.81  4748.6 1722.48  4774.5 1722.12  4834.9 1718.86  4994.3 1718.54
  4994.8 1717.54  5005.2 1717.54  5005.7 1718.54  5113.9 1720.70  5155.6 1719.27
  5205.9 1720.40  5334.8 1719.69  5512.6 1719.46  5536.3 1719.92  5666.0 1719.16
  5708.7 1720.59  5715.4 1722.55  5729.6 1723.90  5751.4 1724.50  5755.2 1726.89
#Mann=12,-1,0
  3971.7    0.12       0  4141.3    0.05       0  4199.8    0.12       0
  4368.8    0.05       0  4426.6    0.12       0  4603.1    0.05       0
  4774.5    0.12       0  4994.3    0.07       0  5005.7    0.12       0
  5334.8    0.05       0  5512.6    0.12       0  5536.3    0.05       0
Bank Sta=4994.3,5005.7
Exp/Cntr=0.3,0.1

Type RM Length L Ch R = 1,84067,767,767,767
BEGIN DESCRIPTION:
Mapping XS 81fed95d
END DESCRIPTION:
XS GIS Cut Line= 3
      1573725.94      6936891.70      1572699.91      6937051.86
      1571623.85      6937572.37
#Sta/Elev= 30
  3966.6 1723.62  4090.4 1721.22  4191.1 1720.51  4291.7 1720.60  4392.6 1719.25
  4433.6 1720.54  4463.5 1719.32  4554.1 1719.31  4559.1 1718.53  4629.8 1719.92
  4757.6 1718.18  4797.5 1718.69  4908.8 1717.85  4951.0 1718.61  4994.3 1717.27
  4994.8 1716.27  5005.2 1716.27  5005.7 1717.27  5070.1 1717.29  5177.1 1718.34
  5277.1 1717.54  5328.1 1718.95  5410.4 1718.14  5508.9 1719.24  5582.2 1717.63
  5932.5 1720.08  6112.9 1719.43  6143.6 1720.99  6188.0 1721.12  6200.4 1723.08
#Mann=8,-1,0
  3966.6    0.12       0  4090.4    0.05       0  4191.1    0.12       0
  4291.7    0.05       0  4629.8    0.12       0  4994.3    0.07       0
  5005.7    0.12       0  5070.1    0.05       0
Bank Sta=4994.3,5005.7
Exp/Cntr=0.3,0.1

Type RM Length L Ch R = 1,83300,348,348,348
BEGIN DESCRIPTION:
Mapping XS f17e2abc
END DESCRIPTION:
XS GIS Cut Line= 3
      1573050.27      6935925.71      1572569.78      6936366.16
      1571613.84      6937432.21
#Sta/Elev= 30
  4356.4 1727.47  4368.8 1727.59  4376.2 1726.27  4382.9 1723.16  4397.1 1721.18
  4485.5 1720.31  4531.5 1721.03  4650.5 1719.46  4714.5 1719.03  4781.8 1718.71
  4878.7 1717.55  4906.5 1718.82  4994.3 1716.90  4994.8 1715.90  5005.7 1716.90
  5161.4 1718.79  5246.6 1717.47  5275.1 1718.86  5296.0 1717.24  5373.7 1716.90
  5586.8 1718.92  5855.9 1717.73  6315.7 1719.33  6351.6 1721.03  6358.3 1724.40
  6365.8 1725.11  6372.5 1727.94  6386.7 1728.99  6400.9 1728.92  6440.1 1722.37
#Mann=7,-1,0
  4356.4    0.05       0  4485.5    0.12       0  4650.5    0.05       0
  4714.5    0.12       0  4781.8    0.05       0  4994.3    0.05       0
  5005.7    0.05       0
Bank Sta=4994.3,5005.7
Exp/Cntr=0.3,0.1

Type RM Length L Ch R = 1,82952,499,499,499
BEGIN DESCRIPTION:
Mapping XS d6a25b5e
END DESCRIPTION:
XS GIS Cut Line= 2
      1572757.94      6935512.11      1571592.67      6937168.98
#Sta/Elev= 30
  4225.8 1722.74  4325.6 1720.09  4539.9 1718.23  4554.7 1717.09  4599.2 1719.11
  4612.0 1717.34  4643.8 1716.51  4809.3 1715.90  4841.1 1716.48  4987.0 1716.09
  4994.3 1715.75  4994.8 1714.75  5005.2 1714.75  5005.7 1715.75  5244.7 1717.21
  5337.1 1715.87  5402.4 1717.74  5503.5 1716.76  5595.8 1719.39  5652.5 1717.50
  5732.6 1718.91  5761.2 1717.33  5854.6 1719.37  6091.3 1719.20  6119.4 1718.24
  6134.2 1719.62  6163.8 1718.95  6169.9 1720.64  6190.9 1721.00  6251.4 1719.24
#Mann=7,-1,0
  4225.8    0.05       0  4643.8    0.12       0  4809.3    0.05       0
  4841.1    0.12       0  4987.0    0.05       0  4994.3    0.05       0
  5005.7    0.05       0
Bank Sta=4994.3,5005.7
Exp/Cntr=0.3,0.1

Type RM Length L Ch R = 1,82453,736,736,736
BEGIN DESCRIPTION:
Mapping XS b77919f8
END DESCRIPTION:
XS GIS Cut Line= 2
      1572219.41      6935004.81      1571513.69      6937101.95
#Sta/Elev= 30
  4121.2 1717.46  4177.1 1716.88  4182.3 1719.07  4208.6 1717.03  4213.8 1719.99
  4240.1 1717.21  4245.3 1719.53  4409.4 1714.55  4662.7 1713.13  4712.6 1711.90
  4757.6 1706.32  4799.8 1706.98  4820.9 1712.02  4989.7 1710.75  4994.3 1706.30
  4994.8 1705.30  5005.7 1706.30  5010.9 1711.11  5027.6 1711.51  5200.8 1711.59
  5431.9 1715.61  5665.0 1717.13  5833.8 1716.25  5846.7 1719.03  5865.5 1718.06
  5873.0 1720.72  5878.2 1717.54  5886.6 1719.19  5904.5 1716.17  6333.9 1718.15
#Mann=3,-1,0
  4121.2    0.05       0  4994.3    0.05       0  5005.7    0.05       0
Bank Sta=4994.3,5005.7
Exp/Cntr=0.3,0.1

Type RM Length L Ch R = 1,81717,606,606,606
BEGIN DESCRIPTION:
Mapping XS 11d614e6
END DESCRIPTION:
XS GIS Cut Line= 3
      1571653.86      6935224.98      1571388.58      6935595.37
      1570993.18      6936751.54
#Sta/Elev= 30
  4130.6 1717.66  4203.9 1717.75  4245.7 1716.41  4260.5 1717.05  4281.9 1715.43
  4310.8 1715.21  4382.1 1716.43  4390.7 1715.78  4417.7 1716.18  4497.5 1715.02
  4518.4 1715.73  4547.9 1715.11  4568.8 1715.75  4645.4 1715.61  4758.1 1714.24
  4884.9 1711.42  4994.3 1710.99  4994.8 1709.99  5005.2 1709.99  5005.7 1710.99
  5085.7 1711.66  5172.2 1711.05  5244.2 1712.66  5328.8 1712.07  5529.6 1715.39
  5599.9 1715.03  5631.2 1716.80  5677.5 1716.73  5709.2 1715.42  5808.1 1715.50
#Mann=3,-1,0
  4130.6    0.05       0  4994.3    0.05       0  5005.7    0.05       0
Bank Sta=4994.3,5005.7
Exp/Cntr=0.3,0.1

Type RM Length L Ch R = 1,81111,1085,1085,1085
BEGIN DESCRIPTION:
Mapping XS f04ea09b
END DESCRIPTION:
XS GIS Cut Line= 3
      1571573.80      6935255.01      1571303.49      6935375.15
      1569968.53      6936035.13
#Sta/Elev= 30
  4247.3 1717.16  4368.6 1714.63  4461.7 1716.72  4597.2 1714.20  4619.5 1714.82
  4649.2 1717.23  4664.1 1716.60  4671.7 1714.94  4694.1 1712.81  4716.5 1711.74
  4798.0 1713.28  4901.6 1711.18  4994.3 1710.89  4994.8 1709.89  5005.2 1709.89
  5005.7 1710.89  5260.6 1712.15  5378.4 1714.99  5485.0 1715.58  5513.0 1716.86
  5535.4 1716.25  5602.8 1717.72  5619.6 1716.84  5634.6 1718.73  5642.1 1717.40
  5670.1 1719.19  5686.9 1717.87  5737.4 1718.19  5880.1 1721.46  6032.3 1723.47
#Mann=3,-1,0
  4247.3    0.05       0  4994.3    0.05       0  5005.7    0.05       0
Bank Sta=4994.3,5005.7
Exp/Cntr=0.3,0.1

Type RM Length L Ch R = 1,80026,759,759,759
BEGIN DESCRIPTION:
Mapping XS 3476cc42
END DESCRIPTION:
XS GIS Cut Line= 3
      1571463.64      6935174.93      1571103.29      6934819.59
      1569811.94      6935189.97
#Sta/Elev= 30
  4318.9 1715.57  4344.1 1715.73  4365.3 1714.06  4400.7 1713.56  4436.0 1709.57
  4485.5 1708.14  4725.9 1706.26  4994.3 1705.95  4994.8 1704.95  5005.2 1704.95
  5005.7 1705.95  5218.5 1706.63  5341.7 1707.95  5395.4 1709.23  5419.5 1710.95
  5426.6 1709.62  5499.4 1709.89  5582.6 1712.62  5598.6 1712.18  5705.1 1714.39
  5728.3 1713.83  5816.7 1715.75  5855.6 1715.55  5923.1 1717.31  5928.3 1716.71
  6034.7 1720.67  6068.5 1721.46  6092.4 1721.01  6134.0 1723.36  6168.4 1723.16
#Mann=3,-1,0
  4318.9    0.05       0  4994.3    0.05       0  5005.7    0.05       0
Bank Sta=4994.3,5005.7
Exp/Cntr=0.3,0.1

Type RM Length L Ch R = 1,79267,824,824,824
BEGIN DESCRIPTION:
Mapping XS a5e50220
END DESCRIPTION:
XS GIS Cut Line= 3
      1571508.73      6935114.92      1570792.97      6934284.04
      1570883.05      6932802.74
#Sta/Elev= 30
  3914.2 1715.77  4000.1 1709.30  4212.9 1706.23  4595.8 1706.20  4729.7 1705.51
  4914.0 1706.10  4992.2 1705.51  4992.7 1704.51  5007.3 1704.51  5007.8 1705.51
  5307.4 1705.79  5608.0 1707.59  5648.1 1706.84  5718.2 1708.43  5828.4 1708.57
  5858.5 1709.36  5938.6 1708.55  5958.6 1709.42  6108.9 1709.99  6129.0 1710.96
  6189.1 1709.30  6219.1 1711.70  6239.2 1715.77  6249.2 1716.22  6259.2 1713.87
  6269.2 1713.07  6282.0 1713.45  6309.3 1712.61  6439.5 1714.75  6494.9 1714.92
#Mann=3,-1,0
  3914.2    0.05       0  4992.2    0.05       0  5007.8    0.05       0
Bank Sta=4992.2,5007.8
Exp/Cntr=0.3,0.1

Type RM Length L Ch R = 1,78443,805,805,805
BEGIN DESCRIPTION:
Mapping XS dea7a2ce
END DESCRIPTION:
XS GIS Cut Line= 2
      1571563.76      6935039.85      1571363.56      6933022.86
#Sta/Elev= 30
  4116.8 1711.53  4159.4 1708.72  4219.1 1707.09  4289.5 1706.15  4462.0 1706.73
  4557.8 1705.87  4663.7 1706.56  4671.4 1706.10  4912.5 1706.15  4992.2 1705.57
  4992.7 1704.57  5007.3 1704.57  5007.8 1705.57  5033.1 1706.09  5053.2 1705.67
  5062.2 1706.23  5143.7 1705.57  5244.2 1706.23  5268.9 1705.73  5495.4 1706.31
  5636.1 1705.84  5786.8 1706.73  5806.9 1707.75  5817.0 1707.48  5857.2 1708.84
  5897.4 1709.14  5980.0 1711.10  6028.0 1713.86  6080.9 1715.32  6143.7 1718.67
#Mann=3,-1,0
  4116.8    0.05       0  4992.2    0.03       0  5007.8    0.05       0
Bank Sta=4992.2,5007.8
Exp/Cntr=0.3,0.1

Type RM Length L Ch R = 1,77638,215,215,215
BEGIN DESCRIPTION:
Mapping XS da46497e
END DESCRIPTION:
XS GIS Cut Line= 2
      1571984.19      6934989.78      1571949.15      6933328.05
#Sta/Elev= 30
  4160.6 1716.61  4192.4 1717.14  4262.4 1715.95  4312.4 1715.98  4322.4 1715.46
  4342.4 1716.18  4352.4 1716.00  4363.3 1715.42  4392.4 1712.42  4402.4 1712.04
  4432.4 1711.39  4452.4 1711.49  4502.5 1709.43  4562.5 1707.92  4592.5 1707.82
  4612.5 1706.94  4772.5 1705.97  4992.2 1705.83  4992.7 1704.83  5007.3 1704.83
  5007.8 1705.83  5322.6 1706.53  5442.7 1708.31  5482.7 1709.90  5602.7 1712.55
  5672.7 1717.10  5682.7 1717.02  5752.7 1719.33  5785.0 1719.59  5822.7 1720.75
#Mann=3,-1,0
  4160.6    0.05       0  4992.2    0.05       0  5007.8    0.05       0
Bank Sta=4992.2,5007.8
Exp/Cntr=0.3,0.1

Type RM Length L Ch R = 1,77423,569,569,569
BEGIN DESCRIPTION:
Mapping XS 4da86e3f
END DESCRIPTION:
XS GIS Cut Line= 2
      1572135.57      6934876.39      1572150.17      6933518.87
#Sta/Elev= 30
  4223.1 1717.48  4241.5 1717.12  4251.5 1715.84  4261.5 1715.62  4281.5 1715.89
  4291.5 1717.09  4311.5 1717.37  4471.5 1716.34  4630.6 1711.75  4635.6 1712.22
  4731.5 1709.12  4811.5 1707.77  4871.5 1707.88  4992.2 1706.88  4992.7 1705.88
  5007.3 1705.88  5007.8 1706.88  5151.5 1708.03  5251.6 1710.06  5321.6 1712.41
  5351.6 1712.60  5361.6 1713.24  5391.6 1713.21  5441.6 1714.96  5461.6 1715.09
  5501.6 1717.32  5521.6 1717.44  5541.6 1716.65  5560.7 1717.20  5580.7 1716.81
#Mann=3,-1,0
  4223.1    0.05       0  4992.2    0.03       0  5007.8    0.05       0
Bank Sta=4992.2,5007.8
Exp/Cntr=0.3,0.1

Type RM Length L Ch R = 1,76854,984,984,984
BEGIN DESCRIPTION:
Mapping XS a8a8eb47
END DESCRIPTION:
XS GIS Cut Line= 2
      1572564.78      6934969.71      1572669.88      6933433.20
#Sta/Elev= 30
  4015.1 1716.31  4056.9 1716.10  4086.8 1715.35  4167.2 1715.70  4227.3 1714.93
  4337.6 1714.50  4407.7 1712.54  4508.0 1711.66  4532.1 1711.86  4548.1 1711.18
  4698.4 1709.92  4778.6 1708.47  4808.7 1708.70  4878.8 1707.96  4979.1 1708.69
  4989.1 1708.61  4992.2 1707.94  4992.7 1706.94  5007.3 1706.94  5007.8 1707.94
  5009.1 1708.55  5059.2 1708.57  5115.9 1709.57  5149.5 1709.19  5159.5 1709.60
  5219.6 1709.75  5239.7 1710.36  5264.3 1710.17  5390.0 1712.22  5555.2 1712.91
#Mann=3,-1,0
  4015.1    0.05       0  4992.2   0.035       0  5007.8    0.05       0
Bank Sta=4992.2,5007.8
Exp/Cntr=0.3,0.1

Type RM Length L Ch R = 1,75870,349,349,349
BEGIN DESCRIPTION:
Mapping XS 34e503ac
END DESCRIPTION:
XS GIS Cut Line= 2
      1573645.87      6934394.15      1572945.19      6933503.28
#Sta/Elev= 30
  4397.3 1714.66  4502.2 1713.72  4587.2 1711.47  4616.1 1711.86  4665.8 1710.21
  4694.7 1710.57  4701.0 1711.61  4709.1 1711.49  4715.5 1710.64  4986.6 1709.25
  4992.2 1707.26  4992.7 1706.26  5007.3 1706.26  5007.8 1707.26  5015.5 1708.92
  5065.2 1708.55  5071.5 1707.75  5086.0 1708.17  5092.3 1707.51  5106.8 1707.26
  5150.1 1708.99  5249.5 1709.71  5264.0 1710.43  5284.8 1710.21  5292.9 1710.82
  5377.9 1710.71  5392.3 1711.28  5485.4 1712.29  5520.6 1713.40  5530.7 1713.10
#Mann=3,-1,0
  4397.3    0.05       0  4992.2    0.03       0  5007.8    0.05       0
Bank Sta=4992.2,5007.8
Exp/Cntr=0.3,0.1

Type RM Length L Ch R = 1,75521,143,143,143
BEGIN DESCRIPTION:
Mapping XS 9b61fd76
END DESCRIPTION:
XS GIS Cut Line= 2
      1573483.38      6934107.55      1573546.64      6933358.21
#Sta/Elev= 30
  4565.0 1711.71  4584.6 1712.03  4614.7 1713.36  4634.8 1713.77  4641.7 1714.57
  4646.8 1714.34  4654.9 1714.59  4664.9 1714.43  4685.0 1715.49  4735.2 1715.11
  4761.4 1713.40  4766.4 1714.99  4785.3 1713.95  4805.4 1713.78  4835.5 1712.87
  4886.1 1712.68  4895.7 1712.90  4935.9 1712.37  4966.0 1712.51  4986.0 1712.16
  4992.2 1710.44  4992.7 1709.44  5007.3 1709.44  5007.8 1710.44  5016.1 1711.98
  5136.6 1710.44  5235.0 1710.92  5277.1 1710.74  5307.2 1712.00  5317.0 1711.37
#Mann=3,-1,0
  4565.0    0.05       0  4992.2    0.03       0  5007.8    0.05       0
Bank Sta=4992.2,5007.8
Exp/Cntr=0.3,0.1

Type RM Length L Ch R = 1,75378,293,293,293
BEGIN DESCRIPTION:
Mapping XS 602b5a74
END DESCRIPTION:
XS GIS Cut Line= 2
      1573570.80      6934053.79      1573680.91      6933318.08
#Sta/Elev= 30
  4544.5 1715.94  4590.8 1716.43  4606.3 1717.15  4621.1 1716.84  4631.2 1717.30
  4670.4 1716.66  4675.5 1717.19  4702.0 1715.48  4712.1 1716.09  4739.6 1716.01
  4744.6 1716.86  4762.7 1715.53  4772.8 1714.33  4793.0 1713.84  4808.8 1710.95
  4823.4 1711.27  4853.7 1710.80  4985.1 1708.47  4992.2 1707.78  4992.7 1706.78
  5007.3 1706.78  5007.8 1707.78  5011.2 1708.15  5080.4 1707.78  5149.6 1708.37
  5207.6 1710.42  5227.8 1709.98  5258.1 1711.69  5268.3 1711.53  5288.4 1709.95
#Mann=3,-1,0
  4544.5    0.05       0  4992.2    0.03       0  5007.8    0.05       0
Bank Sta=4992.2,5007.8
Exp/Cntr=0.3,0.1

Type RM Length L Ch R = 1,75085,357,357,357
BEGIN DESCRIPTION:
Mapping XS 383947ea
END DESCRIPTION:
XS GIS Cut Line= 3
      1575381.03      6933825.37      1573716.94      6933445.84
      1573712.07      6933304.75
#Sta/Elev= 30
  3472.2 1716.14  3531.3 1713.17  3569.2 1712.93  3591.2 1711.62  3652.8 1711.79
  3714.3 1709.54  3775.8 1711.08  3799.6 1710.32  3842.6 1706.81  3847.7 1707.56
  3909.2 1706.38  3928.6 1708.68  3970.7 1704.36  4062.7 1703.49  4237.4 1702.79
  4463.0 1703.79  4534.8 1705.40  4596.4 1704.61  4986.1 1706.62  4992.2 1702.79
  4992.7 1701.79  5007.3 1701.79  5007.8 1702.79  5011.8 1706.64  5017.0 1706.85
  5160.5 1709.22  5226.9 1708.81  5266.9 1711.03  5296.9 1709.74  5320.2 1710.16
#Mann=3,-1,0
  3472.2    0.05       0  4992.2    0.05       0  5007.8    0.05       0
Bank Sta=4992.2,5007.8
Exp/Cntr=0.3,0.1

Type RM Length L Ch R = 1,74728,651,651,651
BEGIN DESCRIPTION:
Mapping XS d8dd14fe
END DESCRIPTION:
XS GIS Cut Line= 2
      1575512.73      6933653.39      1573695.88      6933217.95
#Sta/Elev= 30
  3640.9 1711.47  3710.5 1710.25  3792.8 1710.09  3823.7 1708.92  3864.8 1708.33
  3885.4 1708.23  3900.4 1709.02  3947.6 1706.27  3984.4 1706.02  3989.6 1705.38
  4031.6 1704.32  4068.5 1704.41  4115.6 1703.17  4157.7 1702.78  4546.1 1700.77
  4845.4 1700.16  4965.1 1700.67  4992.2 1700.16  4992.7 1699.16  5007.3 1699.16
  5007.8 1700.16  5013.5 1700.57  5102.6 1700.85  5144.7 1702.01  5170.8 1703.65
  5233.8 1705.64  5317.9 1706.51  5396.8 1708.71  5449.1 1711.33  5509.2 1711.32
#Mann=3,-1,0
  3640.9    0.05       0  4992.2    0.04       0  5007.8    0.05       0
Bank Sta=4992.2,5007.8
Exp/Cntr=0.3,0.1

Type RM Length L Ch R = 1,74077,667,667,667
BEGIN DESCRIPTION:
Mapping XS 266c077f
END DESCRIPTION:
XS GIS Cut Line= 2
      1575007.22      6932887.62      1573807.97      6932787.68
#Sta/Elev= 30
  4444.6 1709.69  4496.1 1707.88  4501.1 1708.47  4507.0 1707.93  4557.2 1706.02
  4607.4 1704.74  4627.4 1704.69  4667.6 1703.81  4828.1 1702.80  4857.3 1702.74
  4862.4 1702.98  4977.7 1702.24  4982.8 1702.55  4991.9 1702.24  4992.4 1701.24
  5007.6 1701.24  5008.1 1702.24  5008.8 1702.46  5038.9 1702.67  5179.4 1702.88
  5209.5 1703.26  5259.6 1705.46  5289.7 1705.79  5344.0 1707.74  5370.0 1708.14
  5470.4 1710.76  5510.5 1710.05  5560.7 1709.80  5600.8 1710.38  5648.0 1709.98
#Mann=3,-1,0
  4444.6    0.05       0  4991.9    0.04       0  5008.1    0.05       0
Bank Sta=4991.9,5008.1
Exp/Cntr=0.3,0.1

Type RM Length L Ch R = 1,73410,657,657,657
BEGIN DESCRIPTION:
Mapping XS 2e13aa99
END DESCRIPTION:
XS GIS Cut Line= 3
      1575234.18      6932589.73      1574760.81      6932298.42
      1573231.36      6931998.00
#Sta/Elev= 30
  4137.1 1710.15  4159.6 1711.71  4253.6 1712.51  4304.5 1710.74  4429.7 1711.42
  4551.8 1710.01  4588.5 1711.18  4594.4 1709.98  4603.9 1710.13  4609.8 1708.89
  4625.2 1708.61  4631.1 1707.49  4698.8 1708.30  4892.5 1702.59  4991.9 1701.49
  4992.4 1700.49  5007.6 1700.49  5008.1 1701.49  5031.2 1702.44  5087.7 1701.75
  5300.1 1702.51  5361.3 1704.29  5575.3 1705.90  5667.0 1708.32  5748.5 1708.09
  5768.9 1709.36  5840.2 1710.15  6093.1 1710.67  6230.0 1710.68  6251.6 1711.27
#Mann=5,-1,0
  4137.1    0.05       0  4991.9    0.05       0  5008.1    0.05       0
  6093.1    0.12       0  6230.0    0.05       0
Bank Sta=4991.9,5008.1
Exp/Cntr=0.3,0.1

Type RM Length L Ch R = 1,72753,624,624,624
BEGIN DESCRIPTION:
Mapping XS f2311981
END DESCRIPTION:
XS GIS Cut Line= 2
      1575373.41      6932594.92      1574141.76      6931111.73
#Sta/Elev= 30
  4130.5 1710.03  4191.5 1710.40  4297.2 1709.04  4311.5 1710.06  4404.0 1709.06
  4432.6 1709.98  4475.6 1708.41  4553.7 1708.06  4617.5 1709.26  4646.2 1707.76
  4808.9 1704.57  4991.9 1702.25  4992.4 1701.25  5007.6 1701.25  5008.1 1702.25
  5220.4 1703.33  5263.4 1704.59  5312.8 1707.42  5391.0 1708.23  5413.1 1710.03
  5448.3 1711.09  5526.4 1709.85  5561.5 1710.24  5596.7 1709.06  5604.5 1709.89
  5717.8 1708.07  5752.9 1708.55  5966.5 1707.25  6023.8 1708.46  6058.4 1708.29
#Mann=3,-1,0
  4130.5    0.05       0  4991.9    0.05       0  5008.1    0.05       0
Bank Sta=4991.9,5008.1
Exp/Cntr=0.3,0.1

Type RM Length L Ch R = 1,72129,1523,1523,1523
BEGIN DESCRIPTION:
Mapping XS cdbe9e7b
END DESCRIPTION:
XS GIS Cut Line= 2
      1575547.03      6932516.81      1574809.77      6930313.70
#Sta/Elev= 30
  3930.7 1707.12  3949.1 1708.99  3980.6 1707.37  4003.3 1708.88  4066.5 1708.06
  4098.2 1706.42  4170.1 1708.54  4224.7 1704.65  4270.1 1704.79  4327.9 1702.41
  4422.7 1701.01  4604.3 1700.03  4927.8 1701.16  4991.9 1700.03  4992.4 1699.03
  5007.6 1699.03  5008.1 1700.03  5131.6 1701.47  5163.2 1703.40  5226.5 1704.83
  5353.0 1703.63  5637.8 1705.00  5690.9 1706.17  5843.5 1705.03  5880.3 1706.22
  6064.5 1706.40  6131.3 1707.79  6143.9 1706.89  6213.1 1707.59  6253.9 1708.53
#Mann=5,-1,0
  3930.7    0.05       0  4991.9    0.05       0  5008.1    0.05       0
  6131.3    0.12       0  6213.1    0.05       0
Bank Sta=4991.9,5008.1
Exp/Cntr=0.3,0.1

Type RM Length L Ch R = 1,70606,593,593,593
BEGIN DESCRIPTION:
Mapping XS 9fd31c70
END DESCRIPTION:
XS GIS Cut Line= 2
      1575859.52      6932560.18      1576276.18      6930537.65
#Sta/Elev= 30
  4159.3 1706.95  4209.3 1706.32  4214.4 1707.19  4233.0 1706.52  4310.0 1707.02
  4396.4 1704.80  4511.2 1703.80  4580.1 1704.43  4672.0 1703.15  4712.9 1703.94
  4774.1 1703.06  4968.1 1703.20  4988.5 1702.97  4991.9 1700.63  4992.4 1699.63
  5007.6 1699.63  5008.1 1700.63  5009.1 1701.84  5070.2 1702.83  5396.3 1700.70
  5529.7 1702.78  5631.8 1702.86  5647.8 1703.91  5723.7 1703.19  5894.2 1704.71
  6019.7 1704.38  6060.6 1705.48  6101.4 1705.22  6162.7 1707.88  6224.3 1706.97
#Mann=3,-1,0
  4159.3    0.05       0  4991.9    0.05       0  5008.1    0.05       0
Bank Sta=4991.9,5008.1
Exp/Cntr=0.3,0.1

Type RM Length L Ch R = 1,70013,2106,2106,2106
BEGIN DESCRIPTION:
Mapping XS 11360e43
END DESCRIPTION:
XS GIS Cut Line= 3
      1576333.43      6932723.67      1576626.40      6931150.35
      1576669.80      6930455.87
#Sta/Elev= 30
  3921.2 1705.58  3937.1 1704.92  3998.2 1705.70  4065.3 1704.18  4110.1 1704.85
  4221.9 1703.51  4354.2 1703.44  4397.0 1704.52  4527.1 1703.17  4618.7 1703.72
  4740.7 1702.41  4811.9 1703.50  4829.1 1702.47  4991.9 1701.86  4992.4 1700.86
  5007.6 1700.86  5008.1 1701.86  5045.2 1703.12  5050.3 1702.56  5127.2 1703.31
  5271.4 1702.28  5624.1 1701.94  5804.5 1703.17  5854.6 1702.62  5964.8 1704.56
  6014.9 1702.87  6095.0 1702.94  6135.1 1704.35  6175.2 1702.81  6217.4 1703.05
#Mann=3,-1,0
  3921.2    0.05       0  4991.9    0.03       0  5008.1    0.05       0
Bank Sta=4991.9,5008.1
Exp/Cntr=0.3,0.1

Type RM Length L Ch R = 1,67907,2212,2212,2212
BEGIN DESCRIPTION:
Mapping XS b70c5d0b
END DESCRIPTION:
XS GIS Cut Line= 3
      1579380.03      6932313.03      1577743.20      6930546.30
      1575677.21      6929652.20
#Sta/Elev= 30
  2947.5 1705.18  2990.1 1704.77  3011.1 1708.79  3039.4 1703.83  3110.3 1700.56
  3273.0 1701.33  3520.7 1697.90  3718.6 1697.76  3817.8 1701.24  3917.0 1697.41
  4179.0 1696.94  4235.7 1699.07  4263.5 1702.75  4313.4 1699.72  4362.7 1700.92
  4398.4 1698.97  4426.6 1699.78  4624.6 1696.88  4991.9 1696.76  4992.4 1695.76
  5008.1 1696.76  5355.9 1698.85  6062.2 1698.67  6091.9 1700.96  6144.4 1700.53
  6167.8 1702.23  6509.0 1700.07  7102.2 1702.90  7324.4 1706.14  7607.1 1705.43
#Mann=3,-1,0
  2947.5    0.05       0  4991.9   0.035       0  5008.1    0.05       0
Bank Sta=4991.9,5008.1
Exp/Cntr=0.3,0.1

Type RM Length L Ch R = 1,65695,964,964,964
BEGIN DESCRIPTION:
Mapping XS 9f18583d
END DESCRIPTION:
XS GIS Cut Line= 3
      1580267.61      6931911.63      1579036.61      6930251.16
      1575790.06      6929270.26
#Sta/Elev= 30
  3116.9 1702.89  3171.2 1703.23  3208.0 1705.94  3228.8 1703.53  3343.6 1701.63
  3585.6 1699.36  3606.9 1701.45  3750.5 1699.04  3930.0 1704.79  4065.6 1703.06
  4229.3 1696.19  4990.3 1695.22  4990.8 1694.22  5009.7 1695.22  5065.1 1696.09
  5138.1 1701.41  5182.8 1696.20  5217.1 1695.43  5519.0 1699.71  5582.6 1697.83
  6533.2 1698.86  7009.3 1696.75  7086.8 1699.95  7151.5 1698.97  7212.2 1701.20
  7306.2 1697.03  7529.7 1696.72  8006.1 1699.56  8258.4 1703.85  8575.4 1704.11
#Mann=3,-1,0
  3116.9    0.05       0  4990.3   0.035       0  5009.7    0.05       0
Bank Sta=4990.3,5009.7
Exp/Cntr=0.3,0.1

Type RM Length L Ch R = 1,64731,1705,1705,1705
BEGIN DESCRIPTION:
Mapping XS 5a3657fe
END DESCRIPTION:
XS GIS Cut Line= 3
      1581411.57      6930596.97      1579816.50      6930108.68
      1576073.05      6928947.67
#Sta/Elev= 30
  3320.1 1702.49  3365.7 1700.91  3540.0 1701.92  3734.8 1696.16  4226.7 1697.14
  4363.0 1694.94  4404.2 1697.54  4799.5 1695.04  4837.5 1697.03  4870.3 1694.89
  4990.3 1694.41  4990.8 1693.41  5009.7 1694.41  5125.9 1694.56  5157.3 1697.26
  5174.6 1694.95  5207.2 1694.51  5510.9 1694.54  6020.6 1696.18  6078.7 1698.17
  6291.8 1696.47  7604.4 1695.69  7659.6 1699.47  7745.2 1696.74  8005.1 1698.60
  8043.7 1700.66  8081.5 1698.69  8282.3 1697.04  8417.8 1699.96  8907.6 1702.66
#Mann=3,-1,0
  3320.1    0.05       0  4990.3    0.05       0  5009.7    0.05       0
Bank Sta=4990.3,5009.7
Exp/Cntr=0.3,0.1

Type RM Length L Ch R = 1,63026,1953,1953,1953
BEGIN DESCRIPTION:
Mapping XS b8676b84
END DESCRIPTION:
XS GIS Cut Line= 3
      1581119.91      6929122.69      1579218.90      6928792.83
      1575948.14      6928385.07
#Sta/Elev= 30
  3352.3 1705.41  3438.5 1702.45  4494.0 1695.96  4813.3 1696.18  4990.3 1693.39
  4990.8 1692.39  5009.7 1693.39  5305.8 1698.24  5366.3 1694.28  5467.0 1693.51
  6900.0 1695.53  7089.5 1699.98  7170.1 1699.21  7217.9 1704.01  7223.0 1701.98
  7260.8 1707.80  7291.1 1706.26  7341.4 1708.46  7371.7 1705.84  7391.8 1708.25
  7432.1 1707.85  7540.8 1702.13  7545.9 1705.11  7613.5 1699.51  7633.7 1702.35
  7702.3 1698.51  7707.3 1701.51  7754.6 1696.76  8348.1 1701.47  8577.8 1700.57
#Mann=3,-1,0
  3352.3    0.05       0  4990.3    0.05       0  5009.7    0.05       0
Bank Sta=4990.3,5009.7
Exp/Cntr=0.3,0.1

Type RM Length L Ch R = 1,61073,1662,1662,1662
BEGIN DESCRIPTION:
Mapping XS 00debe75
END DESCRIPTION:
XS GIS Cut Line= 3
      1581206.71      6926136.60      1578767.51      6927751.16
      1575465.34      6928274.92
#Sta/Elev= 30
  2075.6 1705.37  2149.6 1701.53  2416.4 1703.10  2893.1 1697.93  2936.9 1700.57
  2958.0 1698.59  3102.4 1696.30  3442.4 1696.52  3659.0 1698.74  3788.4 1694.35
  3968.9 1692.62  4104.3 1693.93  4185.5 1691.90  4877.5 1692.11  4989.8 1690.40
  4990.3 1689.40  5010.2 1690.40  5518.9 1691.05  5762.7 1695.81  6198.0 1696.91
  6238.5 1699.17  6268.9 1697.75  6286.7 1699.58  6319.5 1697.94  6608.2 1696.51
  7301.7 1697.26  7463.7 1698.03  7494.0 1701.21  7554.8 1699.12  8344.2 1703.12
#Mann=3,-1,0
  2075.6    0.05       0  4989.8    0.05       0  5010.2    0.05       0
Bank Sta=4989.8,5010.2
Exp/Cntr=0.3,0.1

Type RM Length L Ch R = 1,59411,972,972,972
BEGIN DESCRIPTION:
Mapping XS 005a0262
END DESCRIPTION:
XS GIS Cut Line= 3
      1580199.79      6925173.04      1577491.47      6927212.97
      1575651.21      6927820.60
#Sta/Elev= 30
  2378.3 1700.87  2813.3 1698.50  2871.6 1700.09  3071.5 1696.61  3163.1 1698.87
  3206.8 1695.91  3327.6 1693.60  3492.1 1692.88  3956.4 1696.36  4056.3 1699.69
  4135.4 1705.13  4262.4 1695.52  4476.9 1691.33  4989.8 1689.34  4990.3 1688.34
  5010.2 1689.34  5263.7 1690.81  5370.1 1693.88  5399.2 1696.76  5499.2 1694.88
  5534.6 1697.85  5699.1 1699.59  5975.8 1697.48  6822.5 1698.17  6886.0 1700.95
  6892.0 1703.83  6917.8 1702.88  6923.6 1700.92  7007.7 1700.09  7706.9 1702.47
#Mann=3,-1,0
  2378.3    0.05       0  4989.8   0.035       0  5010.2    0.05       0
Bank Sta=4989.8,5010.2
Exp/Cntr=0.3,0.1

Type RM Length L Ch R = 1,58439,3962,3962,3962
BEGIN DESCRIPTION:
Mapping XS 2ebb1b6b
END DESCRIPTION:
XS GIS Cut Line= 5
      1579904.69      6925173.02      1578316.12      6926067.14
      1576901.19      6926197.34      1575434.17      6926006.37
      1575121.66      6925980.33
#Sta/Elev= 30
  2582.1 1701.00  2865.2 1699.35  2951.9 1704.01  3048.7 1697.79  3121.1 1699.18
  3319.0 1696.34  3415.8 1700.47  3465.3 1695.93  3545.8 1694.40  4465.2 1699.25
  4506.6 1701.77  4684.8 1701.16  4767.6 1696.61  4948.4 1696.90  4986.1 1694.40
  4986.6 1693.40  5013.9 1694.40  5014.2 1696.51  5019.2 1696.67  5179.4 1699.57
  5480.6 1698.18  5852.3 1700.67  6154.9 1698.07  6296.0 1700.41  6507.8 1699.37
  6578.4 1701.70  6840.6 1700.79  7092.7 1703.61  7153.2 1701.56  7618.9 1704.80
#Mann=3,-1,0
  2582.1    0.05       0  4986.1    0.05       0  5013.9    0.05       0
Bank Sta=4986.1,5013.9
Exp/Cntr=0.3,0.1

Type RM Length L Ch R = 1,54477,3855,3855,3855
BEGIN DESCRIPTION:
Mapping XS 55835a42
END DESCRIPTION:
XS GIS Cut Line= 4
      1580555.67      6923914.35      1579166.81      6923662.62
      1578593.90      6923905.68      1574818.91      6925311.53
#Sta/Elev= 30
  3484.6 1701.88  4985.0 1698.58  4986.1 1693.00  4986.6 1692.00  5013.9 1693.00
  5024.0 1699.18  5039.3 1699.77  5306.1 1699.09  5365.2 1701.89  5707.7 1697.91
  5793.3 1700.58  5986.8 1700.16  6146.8 1695.49  6196.7 1696.38  6227.0 1700.52
  6287.6 1695.90  6563.0 1695.80  6600.0 1693.00  6630.3 1694.74  6765.8 1693.64
  6801.6 1695.86  6872.5 1693.50  6967.6 1696.64  6998.0 1694.49  7174.6 1697.62
  7245.9 1695.67  7461.9 1696.55  7511.9 1699.23  7736.8 1695.90  9546.7 1705.08
#Mann=3,-1,0
  3484.6    0.05       0  4986.1    0.03       0  5013.9    0.05       0
Bank Sta=4986.1,5013.9
Exp/Cntr=0.3,0.1

Type RM Length L Ch R = 1,50622,2181,2181,2181
BEGIN DESCRIPTION:
Mapping XS b219fec3
END DESCRIPTION:
XS GIS Cut Line= 3
      1577765.72      6921710.23      1577592.11      6923251.04
      1574955.94      6924943.39
#Sta/Elev= 30
  4922.5 1698.55  4940.4 1699.89  4986.1 1692.25  4986.6 1691.25  5013.9 1692.25
  5171.8 1694.76  5715.3 1692.49  5755.5 1693.04  5836.0 1698.98  5896.4 1695.62
  6097.7 1698.33  6127.8 1696.44  6178.2 1697.42  6409.6 1693.54  6476.1 1695.81
  6497.3 1699.07  6642.6 1693.32  6902.9 1692.25  7017.8 1694.00  7054.2 1696.44
  7547.7 1694.55  7605.2 1699.81  7656.7 1696.29  7871.9 1695.11  8604.0 1697.72
  8770.5 1700.96  9073.1 1699.52  9327.4 1703.23  9415.3 1700.97  9605.7 1705.13
#Mann=3,-1,0
  4922.5    0.05       0  4986.1    0.05       0  5013.9    0.05       0
Bank Sta=4986.1,5013.9
Exp/Cntr=0.3,0.1

Type RM Length L Ch R = 1,48441,2335,2335,2335
BEGIN DESCRIPTION:
Mapping XS 02366807
END DESCRIPTION:
XS GIS Cut Line= 4
      1576614.45      6921753.60      1576848.84      6922864.76
      1576918.28      6923350.87      1574869.85      6924826.43
#Sta/Elev= 30
  3923.8 1697.18  3947.2 1698.67  4173.6 1695.13  4510.8 1697.25  4684.6 1695.72
  4848.1 1696.72  4889.0 1698.71  4985.7 1693.76  4986.2 1692.76  5013.8 1692.76
  5014.3 1693.76  5173.8 1694.38  5194.0 1695.78  5214.2 1694.73  5295.0 1696.79
  5345.5 1695.02  5456.6 1696.97  5586.8 1697.17  5865.4 1695.32  6158.7 1696.72
  6324.4 1695.40  6955.2 1698.50  7192.0 1697.47  7470.6 1700.20  7520.9 1699.25
  7686.6 1700.23  7822.2 1701.36  7849.8 1703.05  7885.4 1701.84  8075.0 1704.35
#Mann=3,-1,0
  3923.8    0.05       0  4985.7    0.03       0  5014.3    0.05       0
Bank Sta=4985.7,5014.3
Exp/Cntr=0.3,0.1

Type RM Length L Ch R = 1,46106,1344,1344,1344
BEGIN DESCRIPTION:
Mapping XS 15cfe02e
END DESCRIPTION:
XS GIS Cut Line= 4
      1575651.18      6921336.26      1575208.48      6922716.44
      1575121.67      6923306.72      1574600.84      6925450.80
#Sta/Elev= 30
  2914.1 1699.99  3080.2 1698.17  3176.6 1700.93  3325.5 1698.16  3535.2 1700.12
  3861.1 1696.29  4375.2 1698.04  4421.3 1700.66  4426.3 1698.94  4597.6 1699.84
  4759.3 1696.73  4910.9 1697.70  4982.1 1696.46  4985.7 1693.53  4986.2 1692.53
  5014.3 1693.53  5043.8 1695.17  5134.0 1693.53  5394.9 1697.08  5640.3 1697.62
  5795.0 1701.62  5984.7 1701.07  6227.3 1707.07  6330.2 1707.73  6422.8 1704.58
  6532.8 1706.47  6699.8 1704.14  6872.0 1706.65  7080.8 1705.12  7166.6 1706.90
#Mann=3,-1,0
  2914.1    0.05       0  4985.7    0.05       0  5014.3    0.05       0
Bank Sta=4985.7,5014.3
Exp/Cntr=0.3,0.1

Type RM Length L Ch R = 1,44762,1581,1581,1581
BEGIN DESCRIPTION:
Mapping XS 54e417ab
END DESCRIPTION:
XS GIS Cut Line= 5
      1575477.55      6921301.54      1575199.80      6921596.65
      1574991.47      6922620.95      1574600.84      6922508.11
      1572951.50      6922343.17
#Sta/Elev= 30
  3044.9 1699.38  3320.0 1698.96  3355.7 1703.68  3450.0 1699.16  3533.2 1697.26
  3655.6 1698.06  3796.9 1694.92  3972.0 1694.77  4063.8 1697.14  4257.7 1698.87
  4559.8 1697.61  4627.0 1699.19  4777.2 1697.00  4866.5 1698.23  4985.7 1694.77
  4986.2 1693.77  5014.3 1694.77  5038.5 1696.31  5078.7 1695.11  5154.2 1696.60
  5269.7 1695.01  5355.2 1698.38  5360.3 1696.92  5420.4 1701.02  5520.9 1698.01
  5621.4 1700.30  5782.2 1699.39  6174.2 1706.66  6345.0 1705.03  6559.6 1705.66
#Mann=3,-1,0
  3044.9    0.05       0  4985.7    0.05       0  5014.3    0.05       0
Bank Sta=4985.7,5014.3
Exp/Cntr=0.3,0.1

Type RM Length L Ch R = 1,43181,823,823,823
BEGIN DESCRIPTION:
Mapping XS 9cd1b707
END DESCRIPTION:
XS GIS Cut Line= 4
      1575413.09      6919963.70      1574720.36      6920474.13
      1574084.95      6921291.84      1572980.78      6922218.93
#Sta/Elev= 30
  2979.5 1701.36  3074.9 1699.91  3138.6 1701.18  3175.1 1699.17  3603.2 1700.57
  3824.6 1697.63  4216.9 1698.40  4351.8 1696.45  4395.2 1698.28  4438.7 1696.54
  4474.0 1698.39  4623.3 1696.01  4702.0 1696.61  4722.8 1699.57  4731.0 1698.07
  4801.6 1698.71  4822.4 1696.76  4858.0 1698.41  4901.6 1696.19  4985.5 1695.57
  4986.0 1694.57  5014.5 1695.57  5214.0 1698.93  5298.5 1702.98  5355.7 1701.50
  5411.7 1706.58  5688.8 1700.81  6164.9 1705.46  6242.9 1703.69  6317.3 1704.35
#Mann=3,-1,0
  2979.5    0.05       0  4985.5    0.05       0  5014.5    0.05       0
Bank Sta=4985.5,5014.5
Exp/Cntr=0.3,0.1
