--- Deadman 59.prj (project) ---

Proj Title=Deadman 59 Base Level Engineering
Current Plan=p01
Default Exp/Contr=0.3,0.1
English Units
Geom File=g01
Flow File=f01
Plan File=p01
Y Axis Title=Elevation
X Axis Title(PF)=Main Channel Distance
X Axis Title(XS)=Station
BEGIN DESCRIPTION:
Deadman 59
END DESCRIPTION:
DSS Export Rating Curves= 0
DSS Export Rating Curve Sorted= 0
DSS Export Volume Flow Curves= 0
DXF OffsetX= 0
DXF OffsetY= 0
DXF ScaleX= 1
DXF ScaleY= 10

--- Deadman 59.p01 (plan) ---

Plan Title=Multiple Run
Short Identifier=Multiple
Geom File=g01
Flow File=f01
Subcritical Flow
K Sum by GR= 0
Std Step Tol= 0.01
Critical Tol= 0.01
Num of Std Step Trials= 20
Max Error Tol= 0.3
Flow Tol Ratio= 0.001
Split Flow NTrial= 30
Split Flow Tol= 0.02
Split Flow Ratio= 0.02
Log Output Level= 0
Friction Slope Method= 1
Unsteady Friction Slope Method= 2
Unsteady Bridges Friction Slope Method= 1
Parabolic Critical Depth
Global Vel Dist=  1 , 1 , 1
Global Log Level= 0
CheckData=True
Encroach Param= -1, 0, 0, 0
BEGIN DESCRIPTION:
Multiple Run
END DESCRIPTION:

--- Deadman 59.f01 (steady flow) ---

Flow Title=Multiple
Number of Profiles=7
Profile Names=10-year,25-year,50-year,1pct_min,100-year,1pct_plu,500-year
River Rch & RM= Deadman 59,Reach-1,17786
     176     237     287     173     344     687     503
River Rch & RM= Deadman 59,Reach-1,17672
     237     326     399     243     485     967     726
River Rch & RM= Deadman 59,Reach-1,11841
     474     672     839     520    1038    2072    1611
River Rch & RM= Deadman 59,Reach-1,2064
     509     728     913     569    1136    2266    1781
Boundary for River Rch & Prof#=Deadman 59,Reach-1,1
Up Type=0
Dn Type=3
Dn Slope=0.007
Boundary for River Rch & Prof#=Deadman 59,Reach-1,2
Up Type=0
Dn Type=3
Dn Slope=0.007
Boundary for River Rch & Prof#=Deadman 59,Reach-1,3
Up Type=0
Dn Type=3
Dn Slope=0.007
Boundary for River Rch & Prof#=Deadman 59,Reach-1,4
Up Type=0
Dn Type=3
Dn Slope=0.007
Boundary for River Rch & Prof#=Deadman 59,Reach-1,5
Up Type=0
Dn Type=3
Dn Slope=0.007
Boundary for River Rch & Prof#=Deadman 59,Reach-1,6
Up Type=0
Dn Type=3
Dn Slope=0.007
Boundary for River Rch & Prof#=Deadman 59,Reach-1,7
Up Type=0
Dn Type=3
Dn Slope=0.007

--- Deadman 59.g01 (geometry) ---

Geom Title=Existing Conditions

River Reach=Deadman 59,Reach-1
Reach XY= 30
      1634805.00      6846788.00      1634258.13      6847539.63
      1634291.78      6847801.67      1634054.51      6848022.80
      1634158.76      6848786.44      1634403.95      6849198.44
      1634357.06      6849982.17      1634653.81      6850098.47
      1634696.92      6850541.31      1634510.35      6850735.27
      1634507.24      6850932.07      1635005.00      6851488.00
      1635221.46      6852455.13      1635856.58      6852834.33
      1636307.44      6852893.52      1636454.63      6853103.27
      1636349.74      6853432.53      1635863.15      6853581.93
      1635656.92      6853899.95      1635571.79      6854371.61
      1635284.87      6854237.59      1635104.91      6854357.88
      1635258.74      6855286.47      1635946.84      6855981.95
      1636303.95      6856848.44      1636302.07      6857080.03
      1636056.54      6857193.85      1636044.64      6857798.16
      1635404.79      6858008.05      1636105.00      6859838.00

Type RM Length L Ch R = 1,17786,114,114,114
BEGIN DESCRIPTION:
Deadman 59 35.0
END DESCRIPTION:
XS GIS Cut Line= 3
      1634555.00      6846688.00      1634755.00      6846838.00
      1634804.99      6846887.99
#Sta/Elev= 30
  4743.8 1891.23  4757.3 1891.13  4771.9 1890.50  4786.5 1890.44  4793.8 1889.92
  4801.1 1889.92  4821.9 1888.98  4836.5 1888.94  4851.1 1888.38  4857.3 1888.50
  4901.1 1887.38  4915.7 1887.46  4921.9 1886.56  4930.3 1887.30  4936.5 1886.95
  4943.8 1887.26  4951.1 1886.42  4957.3 1884.67  4965.7 1880.42  4971.9 1882.30
  4978.3 1879.78  4978.5 1879.28  4982.0 1879.28  4982.3 1879.78  4986.5 1883.83
  4990.7 1880.74  4997.3 1880.74  5036.2 1890.95  5050.4 1891.91  5064.5 1892.15
#Mann=3,-1,0
  4743.8    0.05       0  4978.3    0.05       0  4982.3    0.05       0
Bank Sta=4978.3,4982.3
Exp/Cntr=0.3,0.1

Type RM Length L Ch R = 1,17672,297,297,297
BEGIN DESCRIPTION:
Mapping XS 3557ef7a
END DESCRIPTION:
XS GIS Cut Line= 3
      1634398.62      6846788.10      1634638.23      6846919.81
      1634984.16      6847022.95
#Sta/Elev= 30
  4651.6 1892.94  4826.1 1888.28  4875.7 1887.36  4885.8 1886.82  4891.5 1886.98
  4913.3 1885.94  4920.3 1883.84  4925.0 1883.84  4929.5 1881.73  4929.8 1881.23
  4933.3 1881.23  4933.5 1881.73  4936.8 1881.94  4942.5 1883.15  4953.0 1884.55
  4984.3 1884.89  5008.3 1883.50  5015.6 1883.53  5046.9 1886.52  5074.6 1888.39
  5079.8 1888.32  5107.7 1889.82  5140.8 1891.03  5161.7 1892.42  5172.1 1892.36
  5193.0 1893.79  5203.4 1894.01  5234.7 1895.85  5245.1 1895.80  5286.0 1897.62
#Mann=3,-1,0
  4651.6    0.05       0  4929.5    0.03       0  4933.5    0.05       0
Bank Sta=4929.5,4933.5
Exp/Cntr=0.3,0.1

Type RM Length L Ch R = 1,17375,472,472,472
BEGIN DESCRIPTION:
Deadman 59 34.0
END DESCRIPTION:
XS GIS Cut Line= 3
      1634254.96      6846987.97      1634555.00      6847188.00
      1634805.00      6847188.00
#Sta/Elev= 30
  4633.7 1893.54  4656.3 1892.62  4677.3 1892.29  4683.3 1891.71  4692.3 1891.59
  4705.9 1890.72  4734.4 1889.96  4755.4 1889.04  4806.5 1887.66  4857.6 1886.65
  4863.6 1886.94  4872.6 1886.27  4886.1 1886.12  4908.7 1884.60  4914.7 1884.54
  4922.2 1883.73  4935.7 1883.18  4958.2 1883.27  4971.8 1883.02  4991.3 1881.65
  5034.3 1881.93  5052.3 1881.61  5052.6 1881.11  5056.1 1881.11  5056.3 1881.61
  5084.3 1884.83  5114.3 1885.95  5164.3 1889.78  5224.3 1891.94  5244.3 1893.10
#Mann=3,-1,0
  4633.7    0.05       0  5052.3    0.03       0  5056.3    0.05       0
Bank Sta=5052.3,5056.3
Exp/Cntr=0.3,0.1

Type RM Length L Ch R = 1,16903,448,448,448
BEGIN DESCRIPTION:
Deadman 59 33.0
END DESCRIPTION:
XS GIS Cut Line= 3
      1634055.02      6847488.01      1634255.00      6847538.00
      1634781.33      6847779.21
#Sta/Elev= 30
  4790.3 1890.10  4854.7 1887.16  4862.4 1887.24  4883.0 1886.09  4890.8 1886.20
  4903.7 1884.66  4924.3 1883.85  4944.9 1882.12  4955.2 1881.73  4965.5 1879.33
  4973.2 1879.32  4976.4 1878.98  4976.6 1878.48  4980.1 1878.48  4980.4 1878.98
  4993.9 1879.93  5040.4 1880.99  5062.4 1880.63  5095.4 1879.43  5108.2 1879.41
  5131.2 1880.30  5161.4 1882.38  5251.7 1885.28  5274.7 1885.81  5315.2 1886.12
  5320.7 1886.64  5343.7 1886.46  5381.4 1887.34  5464.2 1888.28  5575.4 1890.42
#Mann=3,-1,0
  4790.3    0.05       0  4976.4    0.05       0  4980.4    0.05       0
Bank Sta=4976.4,4980.4
Exp/Cntr=0.3,0.1

Type RM Length L Ch R = 1,16455,204,204,204
BEGIN DESCRIPTION:
Deadman 59 32.0
END DESCRIPTION:
XS GIS Cut Line= 3
      1633954.99      6847787.99      1634155.00      6847888.00
      1634554.98      6847888.00
#Sta/Elev= 30
  4776.3 1887.70  4821.0 1886.08  4835.0 1885.25  4843.4 1885.16  4874.1 1884.10
  4888.1 1883.15  4896.5 1881.74  4902.1 1881.20  4918.9 1876.98  4924.5 1876.48
  4941.2 1876.55  4944.8 1876.13  4945.1 1875.63  4948.6 1875.63  4948.8 1876.13
  4969.2 1876.25  4991.5 1877.11  5039.9 1877.62  5049.9 1878.22  5069.9 1878.56
  5079.9 1879.48  5089.9 1879.95  5129.9 1881.00  5159.9 1882.08  5199.9 1883.04
  5209.9 1883.58  5219.9 1883.52  5269.9 1884.77  5299.9 1885.80  5399.9 1887.31
#Mann=3,-1,0
  4776.3    0.05       0  4944.8    0.03       0  4948.8    0.05       0
Bank Sta=4944.8,4948.8
Exp/Cntr=0.3,0.1

Type RM Length L Ch R = 1,16251,235,235,235
BEGIN DESCRIPTION:
Mapping XS 59dd8580
END DESCRIPTION:
XS GIS Cut Line= 2
      1633775.74      6847990.69      1634494.51      6848150.42
#Sta/Elev= 30
  4714.4 1890.84  4814.1 1888.03  4826.3 1887.43  4836.6 1886.14  4857.1 1886.38
  4939.0 1882.58  4949.3 1881.58  4955.0 1880.24  4960.1 1879.85  4969.7 1876.86
  4978.0 1874.85  4978.2 1874.35  4981.7 1874.35  4982.0 1874.85  5021.0 1875.21
  5031.2 1875.94  5041.4 1875.90  5047.1 1876.50  5052.3 1876.05  5061.9 1876.27
  5113.2 1877.77  5144.5 1879.21  5164.4 1879.31  5182.9 1880.01  5188.0 1879.50
  5266.8 1881.98  5280.2 1881.93  5323.7 1883.17  5348.8 1883.33  5450.7 1885.50
#Mann=3,-1,0
  4714.4    0.05       0  4978.0    0.03       0  4982.0    0.05       0
Bank Sta=4978,4982
Exp/Cntr=0.3,0.1

Type RM Length L Ch R = 1,16016,260,260,260
BEGIN DESCRIPTION:
Deadman 59 31.0
END DESCRIPTION:
XS GIS Cut Line= 3
      1633754.96      6848137.98      1634055.00      6848288.00
      1634704.96      6848437.99
#Sta/Elev= 30
  4664.8 1889.16  4768.3 1886.68  4880.1 1881.69  4924.8 1878.43  4933.2 1876.98
  4941.6 1874.71  4955.5 1873.93  4977.9 1874.03  4984.2 1873.44  4984.5 1872.94
  4988.0 1872.94  4988.3 1873.44  4991.9 1873.86  5024.2 1873.50  5031.0 1874.03
  5072.1 1873.78  5082.4 1874.29  5102.9 1874.32  5152.5 1877.43  5157.6 1877.22
  5164.5 1878.10  5236.3 1880.25  5248.3 1880.08  5410.8 1883.72  5482.6 1886.39
  5515.1 1887.06  5544.2 1888.43  5636.5 1891.01  5657.1 1891.86  5667.3 1892.77
#Mann=3,-1,0
  4664.8    0.05       0  4984.2    0.05       0  4988.3    0.05       0
Bank Sta=4984.2,4988.3
Exp/Cntr=0.3,0.1

Type RM Length L Ch R = 1,15756,222,222,222
BEGIN DESCRIPTION:
Mapping XS 0dc52cba
END DESCRIPTION:
XS GIS Cut Line= 2
      1633806.99      6848570.55      1634425.06      6848490.69
#Sta/Elev= 30
  4699.4 1885.28  4737.7 1884.09  4755.6 1883.07  4760.6 1883.15  4808.3 1880.36
  4818.4 1879.55  4834.9 1879.26  4840.0 1879.39  4848.6 1878.53  4858.7 1878.10
  4909.1 1874.99  4939.4 1872.34  4949.5 1871.85  4988.6 1871.63  4997.8 1871.37
  4998.1 1870.87  5001.7 1870.87  5001.9 1871.37  5020.0 1871.42  5073.0 1872.59
  5120.9 1875.57  5147.3 1876.79  5221.6 1879.00  5226.6 1878.98  5231.8 1879.75
  5241.9 1879.61  5252.0 1880.29  5262.0 1880.24  5306.0 1881.41  5322.6 1882.38
#Mann=3,-1,0
  4699.4    0.05       0  4997.8    0.03       0  5001.9    0.05       0
Bank Sta=4997.8,5001.9
Exp/Cntr=0.3,0.1

Type RM Length L Ch R = 1,15534,463,463,463
BEGIN DESCRIPTION:
Deadman 59 30.0
END DESCRIPTION:
XS GIS Cut Line= 3
      1633805.00      6848688.00      1634155.00      6848738.00
      1634555.03      6848688.00
#Sta/Elev= 30
  4646.5 1885.61  4697.0 1883.90  4737.4 1881.71  4767.7 1880.84  4798.0 1878.90
  4808.1 1879.07  4838.4 1877.14  4848.5 1876.98  4868.7 1875.35  4899.0 1873.67
  4949.5 1869.24  4977.8 1868.85  4978.0 1868.35  4981.6 1868.35  4981.9 1868.85
  4990.0 1869.19  4997.5 1870.05  5030.3 1870.48  5060.5 1872.74  5090.8 1873.46
  5123.5 1875.03  5161.3 1876.20  5171.4 1877.01  5241.9 1879.81  5262.1 1881.16
  5284.8 1881.85  5292.3 1882.63  5352.8 1884.67  5383.0 1886.64  5403.2 1887.44
#Mann=3,-1,0
  4646.5    0.05       0  4977.8    0.03       0  4981.9    0.05       0
Bank Sta=4977.8,4981.9
Exp/Cntr=0.3,0.1

Type RM Length L Ch R = 1,15071,468,468,468
BEGIN DESCRIPTION:
Deadman 59 29.0
END DESCRIPTION:
XS GIS Cut Line= 3
      1633954.99      6849488.01      1634355.00      6849138.00
      1634555.02      6848937.98
#Sta/Elev= 30
  4468.6 1883.75  4471.9 1883.75  4475.7 1883.04  4490.0 1881.93  4525.1 1880.20
  4539.3 1879.81  4546.9 1880.16  4561.2 1879.62  4574.9 1879.00  4582.0 1878.14
  4667.5 1874.62  4745.3 1872.89  4751.9 1873.26  4759.5 1872.65  4851.6 1870.42
  4886.2 1870.09  4929.4 1869.08  4943.7 1869.17  4991.0 1866.71  4991.2 1866.21
  4994.8 1866.21  4995.1 1866.71  4996.8 1867.13  5014.3 1867.10  5028.4 1867.72
  5042.5 1869.89  5113.3 1875.75  5240.5 1881.30  5254.7 1882.70  5283.0 1883.71
#Mann=3,-1,0
  4468.6    0.05       0  4991.0    0.05       0  4995.1    0.05       0
Bank Sta=4991,4995.1
Exp/Cntr=0.3,0.1

Type RM Length L Ch R = 1,14603,484,484,484
BEGIN DESCRIPTION:
Deadman 59 28.0
END DESCRIPTION:
XS GIS Cut Line= 3
      1634004.99      6849638.00      1634405.00      6849588.00
      1634804.97      6849488.01
#Sta/Elev= 30
  4597.2 1883.07  4627.4 1881.16  4635.0 1880.31  4640.0 1880.43  4647.6 1879.17
  4667.8 1879.41  4738.3 1876.37  4796.2 1871.77  4829.0 1870.64  4876.9 1868.09
  4939.9 1866.81  4957.5 1865.90  4962.5 1866.14  4970.1 1865.34  4995.7 1864.02
  4996.0 1863.52  4999.7 1863.52  5000.0 1864.02  5010.6 1864.24  5018.4 1864.98
  5059.6 1867.10  5064.7 1867.01  5082.8 1868.56  5142.1 1870.59  5229.7 1872.59
  5299.2 1875.64  5353.4 1877.22  5394.6 1880.04  5402.3 1880.90  5412.6 1881.11
#Mann=3,-1,0
  4597.2    0.05       0  4995.7    0.03       0  5000.0    0.05       0
Bank Sta=4995.7,5000
Exp/Cntr=0.3,0.1

Type RM Length L Ch R = 1,14119,459,459,459
BEGIN DESCRIPTION:
Deadman 59 27.0
END DESCRIPTION:
XS GIS Cut Line= 3
      1634005.03      6849938.01      1634405.00      6850038.00
      1634805.01      6849687.99
#Sta/Elev= 30
  4588.7 1882.17  4653.1 1878.64  4660.8 1877.51  4681.4 1877.60  4776.8 1873.86
  4836.1 1871.03  4854.1 1869.22  4900.5 1867.79  4936.6 1865.48  4949.4 1865.26
  4970.1 1862.25  4980.8 1861.78  4981.1 1861.28  4984.8 1861.28  4985.1 1861.78
  4998.4 1863.93  5050.8 1864.98  5100.2 1865.00  5114.4 1864.37  5135.3 1864.56
  5142.9 1863.79  5149.5 1864.36  5157.1 1863.75  5192.2 1865.50  5227.3 1868.15
  5404.8 1873.22  5476.0 1876.72  5525.4 1878.28  5529.2 1879.41  5532.5 1879.41
#Mann=3,-1,0
  4588.7    0.05       0  4980.8    0.05       0  4985.1    0.05       0
Bank Sta=4980.8,4985.1
Exp/Cntr=0.3,0.1

Type RM Length L Ch R = 1,13660,476,476,476
BEGIN DESCRIPTION:
Deadman 59 26.0
END DESCRIPTION:
XS GIS Cut Line= 3
      1633905.04      6850188.00      1634655.00      6850188.00
      1634904.99      6850238.00
#Sta/Elev= 30
  4250.9 1883.23  4280.9 1881.83  4330.9 1880.73  4340.9 1879.98  4350.9 1879.83
  4370.9 1878.10  4410.9 1876.13  4460.9 1874.31  4500.9 1873.54  4530.9 1871.60
  4540.9 1872.27  4700.9 1866.65  4730.9 1865.26  4790.9 1864.22  4830.9 1864.03
  4840.9 1864.37  4910.9 1863.86  4930.9 1863.46  4970.9 1861.04  4978.7 1860.99
  4979.0 1860.49  4982.8 1860.49  4983.1 1860.99  5011.1 1861.20  5031.5 1863.65
  5072.2 1866.27  5113.0 1869.81  5164.0 1871.91  5204.8 1875.93  5255.8 1879.10
#Mann=3,-1,0
  4250.9    0.05       0  4978.7    0.03       0  4983.1    0.05       0
Bank Sta=4978.7,4983.1
Exp/Cntr=0.3,0.1

Type RM Length L Ch R = 1,13184,476,476,476
BEGIN DESCRIPTION:
Deadman 59 25.0
END DESCRIPTION:
XS GIS Cut Line= 3
      1633855.04      6850738.00      1634655.00      6850638.00
      1634954.96      6850438.02
#Sta/Elev= 30
  4192.6 1882.52  4235.4 1881.47  4323.6 1877.46  4515.1 1871.55  4625.9 1867.04
  4646.1 1867.52  4746.8 1865.16  4794.7 1863.19  4799.8 1864.19  4961.0 1859.68
  4988.7 1860.41  5006.3 1858.81  5012.3 1859.16  5019.1 1857.86  5019.4 1857.36
  5023.5 1857.86  5034.8 1857.92  5042.4 1859.99  5048.4 1859.65  5057.4 1861.04
  5063.4 1860.53  5099.4 1862.36  5135.5 1865.02  5150.5 1867.04  5186.6 1869.35
  5207.6 1869.86  5243.7 1872.77  5258.7 1874.85  5315.8 1877.91  5359.3 1881.16
#Mann=3,-1,0
  4192.6    0.05       0  5019.1    0.03       0  5023.5    0.05       0
Bank Sta=5019.1,5023.5
Exp/Cntr=0.3,0.1

Type RM Length L Ch R = 1,12708,237,237,237
BEGIN DESCRIPTION:
Deadman 59 24.0
END DESCRIPTION:
XS GIS Cut Line= 3
      1634305.03      6851137.98      1634555.00      6850988.00
      1634954.99      6850688.01
#Sta/Elev= 30
  4714.5 1871.72  4737.8 1871.07  4772.8 1869.36  4786.4 1868.24  4807.8 1868.03
  4838.9 1866.12  4903.0 1863.96  4947.7 1861.65  4955.5 1859.73  4971.0 1858.46
  4990.2 1855.15  4990.5 1854.65  4994.4 1854.65  4994.7 1855.15  5003.1 1856.32
  5009.1 1856.32  5019.6 1857.71  5034.1 1858.64  5119.6 1858.01  5142.5 1858.20
  5156.0 1857.17  5198.7 1857.76  5227.9 1858.96  5269.6 1859.73  5292.5 1860.90
  5298.7 1860.83  5369.6 1865.94  5377.9 1866.08  5419.6 1868.61  5506.0 1872.10
#Mann=3,-1,0
  4714.5    0.05       0  4990.2    0.05       0  4994.7    0.05       0
Bank Sta=4990.2,4994.7
Exp/Cntr=0.3,0.1

Type RM Length L Ch R = 1,12471,175,175,175
BEGIN DESCRIPTION:
Mapping XS f86ecc61
END DESCRIPTION:
XS GIS Cut Line= 3
      1634393.83      6851317.06      1634827.82      6851108.75
      1634963.21      6850914.34
#Sta/Elev= 30
  4671.5 1870.67  4695.0 1869.87  4702.3 1869.06  4724.9 1869.26  4761.5 1867.80
  4775.7 1867.67  4805.9 1866.13  4843.7 1864.97  4866.3 1863.91  4894.6 1861.44
  4917.2 1859.93  4934.3 1859.23  4950.1 1857.24  4956.9 1855.38  4972.3 1854.74
  4977.3 1854.18  4977.6 1853.68  4981.5 1853.68  4981.8 1854.18  5016.7 1855.33
  5024.9 1856.71  5053.1 1857.87  5166.0 1858.62  5194.1 1859.35  5208.9 1859.28
  5244.7 1859.93  5287.8 1861.56  5301.4 1861.61  5373.2 1863.61  5389.8 1864.44
#Mann=3,-1,0
  4671.5    0.05       0  4977.3    0.03       0  4981.8    0.05       0
Bank Sta=4977.3,4981.8
Exp/Cntr=0.3,0.1

Type RM Length L Ch R = 1,12296,236,236,236
BEGIN DESCRIPTION:
Deadman 59 23.0
END DESCRIPTION:
XS GIS Cut Line= 3
      1634505.02      6851487.99      1634755.00      6851338.00
      1635205.02      6850587.97
#Sta/Elev= 30
  4698.9 1869.86  4733.9 1867.65  4757.2 1868.33  4955.4 1859.71  4976.8 1858.23
  4982.6 1856.84  4987.5 1854.26  4993.3 1854.26  4998.2 1852.62  5001.8 1852.52
  5002.1 1852.02  5006.0 1852.02  5006.3 1852.52  5013.7 1852.70  5025.4 1854.36
  5041.0 1855.35  5083.7 1857.16  5215.9 1858.31  5231.4 1858.83  5258.6 1858.73
  5449.1 1863.61  5538.5 1868.56  5565.7 1869.22  5618.2 1871.40  5655.2 1873.87
  5725.1 1877.45  5756.2 1878.98  5771.8 1879.13  5799.0 1881.13  5865.1 1884.71
#Mann=3,-1,0
  4698.9    0.05       0  5001.8    0.05       0  5006.3    0.05       0
Bank Sta=5001.8,5006.3
Exp/Cntr=0.3,0.1

Type RM Length L Ch R = 1,12060,219,219,219
BEGIN DESCRIPTION:
Mapping XS 028a6011
END DESCRIPTION:
XS GIS Cut Line= 3
      1634657.08      6851593.88      1634930.67      6851503.84
      1635120.42      6850924.23
#Sta/Elev= 30
  4678.2 1865.09  4686.5 1864.20  4712.9 1864.14  4744.7 1862.52  4750.0 1862.83
  4776.5 1861.47  4855.0 1859.26  4928.7 1855.00  4949.7 1852.68  4970.1 1852.21
  4970.4 1851.71  4974.3 1851.71  4974.6 1852.21  5003.9 1852.40  5029.3 1854.44
  5046.0 1854.65  5077.6 1853.36  5124.9 1853.56  5289.4 1855.94  5316.0 1857.28
  5321.2 1856.88  5347.8 1858.14  5361.7 1858.08  5379.7 1859.35  5384.9 1858.96
  5411.5 1860.28  5424.8 1860.27  5443.4 1861.58  5466.9 1862.06  5576.1 1867.38
#Mann=3,-1,0
  4678.2    0.05       0  4970.1    0.05       0  4974.6    0.05       0
Bank Sta=4970.1,4974.6
Exp/Cntr=0.3,0.1

Type RM Length L Ch R = 1,11841,457,457,457
BEGIN DESCRIPTION:
Deadman 59 22.0
END DESCRIPTION:
XS GIS Cut Line= 3
      1634655.01      6851638.00      1635005.00      6851638.00
      1635554.99      6851738.00
#Sta/Elev= 30
  4650.4 1864.95  4670.4 1864.39  4720.4 1861.26  4740.4 1861.60  4760.4 1861.27
  4890.4 1855.82  4900.4 1855.78  4930.4 1854.51  4940.4 1854.56  4960.4 1852.88
  4986.7 1849.48  4987.2 1848.98  4993.5 1848.98  4994.0 1849.48  5002.9 1849.65
  5010.6 1850.70  5020.7 1851.26  5041.1 1851.57  5051.2 1852.78  5061.4 1853.08
  5102.0 1853.06  5138.9 1854.31  5192.2 1855.29  5295.1 1856.15  5362.5 1857.51
  5376.5 1857.22  5407.0 1859.01  5420.9 1859.21  5474.3 1862.33  5559.4 1864.68
#Mann=3,-1,0
  4650.4    0.05       0  4986.7    0.05       0  4994.0    0.05       0
Bank Sta=4986.7,4994
Exp/Cntr=0.3,0.1

Type RM Length L Ch R = 1,11384,449,449,449
BEGIN DESCRIPTION:
Deadman 59 21.0
END DESCRIPTION:
XS GIS Cut Line= 3
      1634650.21      6852057.87      1635155.00      6852038.00
      1635505.01      6851838.00
#Sta/Elev= 30
  4495.3 1865.82  4520.1 1864.74  4550.1 1862.20  4580.2 1860.80  4660.2 1858.63
  4710.3 1858.14  4770.3 1855.47  4860.4 1853.48  4874.4 1852.88  4910.4 1849.99
  4930.4 1849.87  4940.4 1850.74  4980.5 1850.07  4990.5 1849.66  4998.0 1848.30
  5010.5 1847.87  5011.0 1847.37  5017.3 1847.37  5017.8 1847.87  5023.5 1847.88
  5030.0 1849.13  5045.8 1850.91  5051.6 1850.84  5058.1 1851.83  5067.4 1852.20
  5250.3 1854.71  5299.9 1859.59  5330.9 1861.71  5352.5 1862.61  5403.6 1863.45
#Mann=3,-1,0
  4495.3    0.05       0  5010.5    0.05       0  5017.8    0.05       0
Bank Sta=5010.5,5017.8
Exp/Cntr=0.3,0.1

Type RM Length L Ch R = 1,10935,444,444,444
BEGIN DESCRIPTION:
Deadman 59 20.0
END DESCRIPTION:
XS GIS Cut Line= 3
      1635104.99      6852538.01      1635205.00      6852438.00
      1635626.67      6851985.16
#Sta/Elev= 30
  4853.4 1864.42  4857.0 1864.42  4881.7 1860.72  4924.1 1856.24  4966.6 1850.38
  4980.7 1848.07  4991.3 1846.87  4998.3 1846.87  5005.1 1846.44  5005.6 1845.94
  5012.0 1845.94  5012.5 1846.44  5030.3 1847.14  5058.6 1849.16  5072.8 1849.30
  5086.9 1848.66  5093.8 1847.91  5107.9 1848.03  5172.0 1851.20  5327.3 1851.69
  5426.5 1853.16  5454.8 1853.89  5475.8 1855.28  5490.0 1855.78  5497.3 1856.53
  5504.2 1856.53  5511.5 1857.15  5546.7 1858.76  5603.4 1861.14  5613.6 1861.06
#Mann=3,-1,0
  4853.4    0.05       0  5005.1    0.05       0  5012.5    0.05       0
Bank Sta=5005.1,5012.5
Exp/Cntr=0.3,0.1

Type RM Length L Ch R = 1,10491,279,279,279
BEGIN DESCRIPTION:
Deadman 59 19.0
END DESCRIPTION:
XS GIS Cut Line= 3
      1635354.98      6852838.02      1635555.00      6852638.00
      1636204.97      6851838.03
#Sta/Elev= 30
  4716.3 1864.97  4758.8 1862.31  4829.5 1860.34  4886.0 1854.96  4942.6 1847.43
  5002.4 1848.90  5006.4 1850.39  5012.8 1847.81  5020.7 1849.88  5027.2 1848.05
  5035.1 1850.41  5041.5 1848.61  5049.5 1849.43  5055.9 1847.10  5070.3 1848.73
  5105.5 1849.65  5119.8 1846.97  5198.1 1846.33  5212.5 1847.78  5243.9 1846.15
  5244.4 1845.65  5251.4 1846.15  5255.6 1848.39  5262.1 1848.74  5383.5 1850.80
  5411.5 1852.90  5517.8 1856.54  5596.1 1861.65  5866.2 1868.26  6029.9 1874.51
#Mann=3,-1,0
  4716.3    0.05       0  5243.9    0.05       0  5251.4    0.05       0
Bank Sta=5243.9,5251.4
Exp/Cntr=0.3,0.1

Type RM Length L Ch R = 1,10212,626,626,626
BEGIN DESCRIPTION:
Mapping XS 019cfd76
END DESCRIPTION:
XS GIS Cut Line= 2
      1635661.15      6852910.84      1636115.55      6852442.56
#Sta/Elev= 30
  4829.6 1856.07  4841.4 1855.76  4862.5 1853.92  4905.0 1851.85  4912.2 1850.85
  4919.1 1850.64  4926.3 1849.75  4982.9 1845.65  5000.2 1843.13  5000.7 1842.63
  5007.2 1842.63  5007.7 1843.13  5025.3 1845.56  5046.4 1845.46  5053.6 1844.78
  5060.6 1845.63  5067.8 1845.88  5074.7 1845.46  5103.0 1846.48  5216.2 1847.17
  5244.5 1847.82  5265.6 1847.51  5286.9 1848.28  5301.1 1848.16  5315.2 1847.16
  5350.5 1848.90  5421.2 1850.12  5456.7 1851.57  5477.8 1851.57  5482.1 1852.06
#Mann=3,-1,0
  4829.6    0.05       0  5000.2    0.03       0  5007.7    0.05       0
Bank Sta=5000.2,5007.7
Exp/Cntr=0.3,0.1

Type RM Length L Ch R = 1,9586,491,491,491
BEGIN DESCRIPTION:
Mapping XS 2641436b
END DESCRIPTION:
XS GIS Cut Line= 3
      1635598.95      6852930.47      1636062.97      6853058.60
      1636691.60      6852730.47
#Sta/Elev= 30
  4212.3 1859.25  4270.4 1857.58  4331.0 1854.58  4410.1 1852.83  4484.0 1847.86
  4557.8 1845.66  4654.3 1845.07  4671.3 1844.01  4685.4 1844.44  4692.1 1845.34
  4792.0 1844.93  4830.6 1844.19  4932.9 1844.93  4996.6 1842.71  4997.1 1842.21
  5003.9 1842.21  5004.4 1842.71  5067.9 1850.16  5139.8 1853.31  5192.3 1856.74
  5237.4 1860.81  5244.6 1862.08  5260.0 1863.10  5266.6 1864.14  5305.1 1866.69
  5310.8 1867.82  5332.9 1869.06  5339.0 1870.28  5361.5 1871.72  5402.8 1872.20
#Mann=3,-1,0
  4212.3    0.05       0  4996.6    0.03       0  5004.4    0.05       0
Bank Sta=4996.6,5004.4
Exp/Cntr=0.3,0.1

Type RM Length L Ch R = 1,9095,577,577,577
BEGIN DESCRIPTION:
Deadman 59 18.0
END DESCRIPTION:
XS GIS Cut Line= 3
      1635554.95      6852987.98      1636355.00      6853338.00
      1636704.98      6853288.00
#Sta/Elev= 30
  4120.8 1860.64  4187.5 1858.44  4251.8 1857.65  4339.2 1853.84  4385.5 1853.28
  4502.5 1845.94  4531.3 1845.02  4583.6 1843.84  4659.2 1843.56  4682.6 1842.44
  4706.0 1844.09  4797.6 1842.32  4819.4 1840.42  4833.8 1840.55  4851.8 1842.19
  4857.2 1841.67  4863.1 1842.76  4961.7 1843.10  4979.6 1842.68  5020.5 1839.80
  5021.0 1839.30  5028.3 1839.80  5034.5 1840.97  5074.9 1841.24  5105.2 1846.50
  5155.7 1851.38  5206.2 1855.03  5297.1 1864.05  5317.3 1867.13  5347.6 1869.96
#Mann=3,-1,0
  4120.8    0.05       0  5020.5    0.05       0  5028.3    0.05       0
Bank Sta=5020.5,5028.3
Exp/Cntr=0.3,0.1

Type RM Length L Ch R = 1,8518,386,386,386
BEGIN DESCRIPTION:
Deadman 59 17.0
END DESCRIPTION:
XS GIS Cut Line= 3
      1635704.97      6853287.97      1635934.85      6853515.68
      1636405.01      6853888.01
#Sta/Elev= 30
  4682.1 1854.84  4724.5 1852.44  4781.1 1850.13  4802.3 1848.28  4844.8 1846.02
  4851.8 1846.06  4873.1 1844.27  4922.5 1842.50  4936.7 1841.27  4957.9 1838.04
  4972.1 1837.58  4975.1 1836.97  4975.6 1836.47  4982.5 1836.47  4983.0 1836.97
  5003.8 1838.42  5085.3 1840.60  5120.7 1840.98  5135.0 1840.14  5143.1 1840.26
  5149.4 1841.25  5235.5 1841.88  5242.4 1842.34  5263.2 1842.22  5341.7 1843.84
  5413.9 1845.94  5426.8 1845.94  5527.7 1849.93  5541.6 1850.16  5605.4 1855.09
#Mann=3,-1,0
  4682.1    0.05       0  4975.1    0.03       0  4983.0    0.05       0
Bank Sta=4975.1,4983
Exp/Cntr=0.3,0.1

Type RM Length L Ch R = 1,8132,350,350,350
BEGIN DESCRIPTION:
Deadman 59 16.0
END DESCRIPTION:
XS GIS Cut Line= 3
      1635354.96      6853587.98      1635744.40      6853837.71
      1636505.04      6854138.01
#Sta/Elev= 30
  4564.5 1853.39  4666.0 1849.67  4759.8 1847.47  4890.0 1842.42  4962.7 1838.97
  4977.9 1838.76  5000.9 1836.10  5001.4 1835.60  5008.5 1835.60  5009.0 1836.10
  5024.5 1836.93  5060.0 1836.85  5091.5 1838.55  5135.3 1839.24  5150.9 1838.51
  5175.3 1839.78  5337.6 1842.54  5350.3 1843.27  5421.5 1844.46  5475.6 1846.49
  5529.7 1849.03  5597.6 1855.15  5651.3 1858.93  5683.6 1863.02  5697.4 1863.37
  5751.5 1866.82  5791.1 1868.44  5800.2 1869.45  5805.6 1869.28  5844.9 1872.18
#Mann=3,-1,0
  4564.5    0.05       0  5000.9    0.05       0  5009.0    0.05       0
Bank Sta=5000.9,5009
Exp/Cntr=0.3,0.1

Type RM Length L Ch R = 1,7782,278,278,278
BEGIN DESCRIPTION:
Deadman 59 15.0
END DESCRIPTION:
XS GIS Cut Line= 3
      1635254.99      6853737.99      1635655.00      6854138.00
      1636054.99      6854337.99
#Sta/Elev= 30
  4435.5 1853.20  4548.6 1848.96  4661.8 1845.90  4704.2 1844.28  4732.5 1842.99
  4760.8 1841.06  4803.2 1838.91  4845.6 1838.06  4944.6 1837.50  4972.9 1836.59
  4987.1 1835.69  5023.6 1835.44  5027.9 1835.10  5028.4 1834.60  5035.5 1834.60
  5036.0 1835.10  5059.9 1835.95  5082.3 1838.24  5104.6 1838.17  5113.0 1838.95
  5121.4 1839.22  5135.4 1839.06  5188.5 1840.47  5194.1 1840.32  5238.8 1841.12
  5291.9 1842.82  5328.2 1845.40  5381.3 1851.07  5389.7 1851.30  5448.4 1855.49
#Mann=3,-1,0
  4435.5    0.05       0  5027.9    0.03       0  5036.0    0.05       0
Bank Sta=5027.9,5036
Exp/Cntr=0.3,0.1

Type RM Length L Ch R = 1,7504,386,386,386
BEGIN DESCRIPTION:
Mapping XS 60c22960
END DESCRIPTION:
XS GIS Cut Line= 3
      1635268.77      6854039.27      1635501.43      6854317.08
      1635650.37      6854466.02
#Sta/Elev= 30
  4550.8 1844.93  4646.6 1841.24  4660.9 1839.65  4675.2 1839.13  4681.7 1839.86
  4731.8 1838.02  4745.5 1836.65  4777.4 1835.29  4810.0 1836.12  4866.5 1836.00
  4874.3 1837.73  4888.3 1839.32  4895.1 1838.78  4909.4 1835.85  4923.4 1834.89
  4930.5 1835.76  4937.6 1835.07  4944.6 1835.63  4951.7 1833.89  4958.8 1834.35
  4965.8 1832.85  4983.0 1832.48  4983.5 1831.98  4991.1 1832.48  5015.3 1837.20
  5036.5 1836.14  5071.9 1837.07  5079.0 1836.22  5100.2 1837.92  5123.8 1838.66
#Mann=3,-1,0
  4550.8    0.05       0  4983.0    0.03       0  4991.1    0.05       0
Bank Sta=4983,4991.1
Exp/Cntr=0.3,0.1

Type RM Length L Ch R = 1,7118,213,213,213
BEGIN DESCRIPTION:
Mapping XS bf6ff628
END DESCRIPTION:
XS GIS Cut Line= 3
      1635154.21      6854115.69      1635352.53      6854429.70
      1635651.04      6854608.78
#Sta/Elev= 30
  4837.6 1845.68  4905.0 1843.57  4926.2 1841.67  4956.7 1838.00  4970.4 1833.54
  4979.8 1831.30  4980.3 1830.80  4987.5 1830.80  4988.0 1831.30  4993.2 1831.32
  5020.3 1836.53  5029.6 1835.74  5035.6 1834.38  5065.1 1835.35  5129.7 1835.87
  5159.7 1836.00  5166.2 1835.00  5195.2 1836.34  5212.2 1835.94  5253.5 1837.19
  5327.3 1836.29  5333.2 1835.82  5340.1 1834.23  5348.7 1833.76  5363.5 1835.88
  5370.1 1835.81  5375.9 1834.56  5444.0 1834.42  5538.4 1840.95  5557.1 1843.59
#Mann=3,-1,0
  4837.6    0.05       0  4979.8    0.05       0  4988.0    0.05       0
Bank Sta=4979.8,4988
Exp/Cntr=0.3,0.1

Type RM Length L Ch R = 1,6905,149,149,149
BEGIN DESCRIPTION:
Deadman 59 14.0
END DESCRIPTION:
XS GIS Cut Line= 4
      1634841.69      6854351.80      1635105.00      6854388.00
      1635337.32      6854459.90      1635578.08      6854588.64
#Sta/Elev= 30
  4734.2 1846.58  4899.1 1842.40  4929.3 1840.02  4949.5 1837.30  4964.0 1833.74
  4969.7 1831.66  4993.3 1830.21  4993.8 1829.71  5001.1 1829.71  5001.6 1830.21
  5010.5 1830.65  5021.5 1834.44  5054.1 1837.63  5062.8 1837.87  5073.3 1836.98
  5081.5 1833.89  5086.8 1833.82  5198.9 1835.94  5308.1 1836.80  5352.0 1836.40
  5365.3 1835.63  5374.0 1833.73  5388.0 1835.08  5401.6 1834.34  5417.9 1835.34
  5456.0 1833.75  5461.8 1834.27  5478.0 1833.51  5500.0 1835.97  5516.2 1836.71
#Mann=3,-1,0
  4734.2    0.05       0  4993.3    0.05       0  5001.6    0.05       0
Bank Sta=4993.3,5001.6
Exp/Cntr=0.3,0.1

Type RM Length L Ch R = 1,6756,159,159,159
BEGIN DESCRIPTION:
Mapping XS 8c6d95fc
END DESCRIPTION:
XS GIS Cut Line= 4
      1634796.46      6854556.15      1635313.65      6854524.18
      1635388.98      6854525.12      1635569.27      6854601.97
#Sta/Elev= 30
  4690.4 1846.31  4729.0 1844.47  4859.3 1842.00  4898.9 1839.60  4929.4 1839.51
  4959.5 1837.10  4979.5 1832.83  4989.5 1829.98  5005.4 1829.52  5005.9 1829.02
  5013.2 1829.02  5013.7 1829.52  5029.6 1832.20  5049.6 1833.06  5059.6 1832.31
  5065.1 1832.63  5070.1 1833.90  5079.7 1832.87  5099.7 1834.78  5283.9 1836.45
  5299.9 1836.31  5312.2 1834.22  5323.1 1833.92  5358.1 1834.26  5376.2 1835.86
  5388.3 1834.57  5399.2 1834.66  5434.4 1833.02  5458.0 1834.19  5479.9 1836.15
#Mann=3,-1,0
  4690.4    0.05       0  5005.4    0.05       0  5013.7    0.05       0
#XS Ineff=2,0
       0                 5240.30    0.00 1840.64
Permanent Ineff=
       F       F
Bank Sta=5005.4,5013.7
Exp/Cntr=0.3,0.1

Type RM Length L Ch R = 1,6597,127,127,127
BEGIN DESCRIPTION:
Mapping XS b45a237d
END DESCRIPTION:
XS GIS Cut Line= 4
      1634632.89      6854824.58      1635155.74      6854682.61
      1635369.58      6854619.04      1635584.05      6854624.13
#Sta/Elev= 30
  4509.8 1851.63  4657.1 1844.96  4819.4 1840.81  4833.2 1841.59  4859.2 1838.51
  4864.4 1839.55  4885.0 1837.02  4905.7 1836.52  4957.6 1831.00  4978.6 1827.46
  5008.1 1827.36  5009.1 1825.58  5009.6 1825.08  5017.4 1825.58  5047.9 1826.85
  5050.8 1825.92  5092.5 1826.04  5134.3 1833.79  5165.6 1837.57  5185.9 1836.27
  5191.1 1837.16  5196.9 1835.62  5217.7 1834.93  5280.1 1835.89  5360.1 1835.21
  5380.1 1831.43  5410.1 1833.45  5430.1 1831.67  5450.1 1834.74  5489.2 1838.20
#Mann=3,-1,0
  4509.8    0.05       0  5009.1    0.05       0  5017.4    0.05       0
#XS Ineff=2,0
       0                 5161.60    0.00 1844.37
Permanent Ineff=
       F       F
Bank Sta=5009.1,5017.4
Exp/Cntr=0.3,0.1

Type RM Length L Ch R = 1,6470,195,195,195
BEGIN DESCRIPTION:
Deadman 59 13.0
END DESCRIPTION:
XS GIS Cut Line= 4
      1634608.67      6855001.17      1635141.89      6854810.73
      1635421.57      6854730.27      1635747.52      6854636.51
#Sta/Elev= 30
  4444.8 1858.63  4524.5 1850.27  4586.1 1847.65  4616.9 1845.40  4844.4 1839.00
  4929.4 1838.00  4950.6 1836.67  4975.8 1833.69  4982.5 1830.34  4988.9 1829.58
  4989.4 1829.08  4997.2 1829.58  5006.6 1830.91  5034.4 1831.44  5055.9 1833.97
  5118.3 1833.23  5184.8 1833.74  5191.1 1832.18  5211.9 1832.49  5223.7 1833.22
  5232.8 1834.95  5243.2 1835.18  5336.8 1834.62  5402.6 1830.47  5420.1 1833.88
  5441.5 1835.07  5470.0 1838.75  5524.1 1843.47  5586.6 1845.22  5641.2 1848.22
#Mann=3,-1,0
  4444.8    0.05       0  4988.9    0.05       0  4997.2    0.05       0
#XS Ineff=2,0
    0.00 4753.10 1840.76 5246.90    0.00 1840.76
Permanent Ineff=
       F       F
Bank Sta=4988.9,4997.2
Exp/Cntr=0.3,0.1

Type RM Length L Ch R = 1,6275,134,134,134
BEGIN DESCRIPTION:
Mapping XS e0da5233
END DESCRIPTION:
XS GIS Cut Line= 3
      1634849.41      6855074.59      1635277.23      6854968.61
      1635711.46      6854835.61
#Sta/Elev= 30
  4639.5 1844.10  4725.9 1840.57  4830.7 1837.76  4850.1 1836.42  4902.8 1835.63
  4938.1 1833.07  4954.3 1831.40  4975.3 1828.41  4975.8 1827.91  4983.1 1827.91
  4983.6 1828.41  4995.5 1829.50  5020.9 1829.75  5047.1 1832.63  5076.5 1834.54
  5096.5 1833.72  5119.8 1833.92  5151.1 1832.42  5200.0 1831.74  5224.3 1831.91
  5265.5 1833.76  5308.8 1833.45  5328.9 1832.61  5349.8 1829.41  5401.8 1832.45
  5412.6 1833.87  5445.0 1836.46  5505.3 1840.58  5510.6 1841.43  5534.4 1842.72
#Mann=3,-1,0
  4639.5    0.05       0  4975.3    0.05       0  4983.6    0.05       0
#XS Ineff=2,0
       0                 5073.10    0.00 1837.58
Permanent Ineff=
       F       F
Bank Sta=4975.3,4983.6
Exp/Cntr=0.3,0.1

Type RM Length L Ch R = 1,6141,182,182,182
BEGIN DESCRIPTION:
Mapping XS 07aebb77
END DESCRIPTION:
XS GIS Cut Line= 4
      1634987.58      6855185.12      1635321.66      6855085.89
      1635490.94      6855027.53      1635777.24      6854928.82
#Sta/Elev= 30
  4746.0 1840.00  4855.8 1835.24  4894.3 1834.33  4932.7 1832.40  4965.9 1829.90
  4972.8 1828.55  4994.9 1828.08  4995.4 1827.58  5003.3 1828.08  5014.5 1828.20
  5045.8 1832.53  5065.5 1832.17  5087.6 1833.55  5140.3 1833.36  5182.7 1830.66
  5235.5 1833.31  5267.3 1833.46  5299.0 1832.31  5321.8 1832.64  5353.0 1831.07
  5373.1 1828.24  5378.9 1830.12  5394.2 1831.00  5410.1 1830.44  5415.4 1828.48
  5447.1 1830.65  5467.3 1831.19  5478.8 1833.61  5503.7 1835.48  5576.4 1836.84
#Mann=3,-1,0
  4746.0    0.05       0  4994.9    0.03       0  5003.3    0.05       0
#XS Ineff=2,0
       0                 5088.20    0.00 1835.70
Permanent Ineff=
       F       F
Bank Sta=4994.9,5003.3
Exp/Cntr=0.3,0.1

Type RM Length L Ch R = 1,5959,436,436,436
BEGIN DESCRIPTION:
Deadman 59 12.0
END DESCRIPTION:
XS GIS Cut Line= 4
      1634854.97      6855438.01      1635255.00      6855288.00
      1635574.35      6855150.41      1635875.61      6855020.62
#Sta/Elev= 30
  4568.7 1857.89  4600.8 1855.00  4608.8 1853.49  4632.8 1851.98  4644.4 1850.14
  4675.5 1847.53  4815.3 1839.81  4846.4 1837.47  4865.1 1837.05  4878.5 1835.96
  4920.3 1834.27  4963.9 1830.92  4974.6 1829.73  4989.1 1826.93  4989.6 1826.43
  4997.0 1826.43  4997.5 1826.93  5028.5 1827.73  5050.4 1830.48  5062.9 1829.74
  5086.4 1830.90  5104.5 1830.36  5180.5 1832.11  5246.4 1832.93  5443.0 1832.65
  5537.1 1828.32  5542.6 1829.18  5560.6 1829.46  5642.1 1835.30  5671.7 1836.25
#Mann=3,-1,0
  4568.7    0.05       0  4989.1    0.03       0  4997.5    0.05       0
#XS Ineff=2,0
       0                 5251.40    0.00 1836.27
Permanent Ineff=
       F       F
Bank Sta=4989.1,4997.5
Exp/Cntr=0.3,0.1

Type RM Length L Ch R = 1,5523,495,495,495
BEGIN DESCRIPTION:
Deadman 59 11.0
END DESCRIPTION:
XS GIS Cut Line= 4
      1635354.96      6855738.03      1635555.00      6855588.00
      1635751.43      6855254.58      1635905.27      6854993.45
#Sta/Elev= 30
  4750.4 1840.55  4836.9 1835.61  4850.4 1834.42  4857.7 1832.79  4864.0 1832.39
  4893.2 1832.76  4914.0 1830.50  4936.9 1829.09  4957.7 1826.28  4986.9 1825.85
  4993.1 1824.82  4993.6 1824.32  5001.0 1824.32  5001.5 1824.82  5014.1 1824.99
  5029.7 1826.89  5035.5 1828.38  5045.4 1828.69  5072.6 1828.30  5116.5 1829.49
  5174.5 1829.76  5264.0 1829.28  5328.4 1831.36  5445.5 1830.83  5476.3 1830.08
  5519.7 1827.88  5599.7 1833.41  5605.5 1834.36  5627.2 1835.95  5690.5 1837.38
#Mann=3,-1,0
  4750.4    0.05       0  4993.1    0.05       0  5001.5    0.05       0
#XS Ineff=2,0
       0                 5366.30    0.00 1833.16
Permanent Ineff=
       F       F
Bank Sta=4993.1,5001.5
Exp/Cntr=0.3,0.1

Type RM Length L Ch R = 1,5028,470,470,470
BEGIN DESCRIPTION:
Deadman 59 10.0
END DESCRIPTION:
XS GIS Cut Line= 3
      1635504.99      6856088.00      1635905.00      6855938.00
      1636305.00      6855538.00
#Sta/Elev= 30
  4574.3 1839.58  4614.4 1837.31  4638.4 1836.83  4681.1 1834.27  4705.1 1833.37
  4713.2 1832.08  4723.8 1831.90  4735.4 1832.42  4745.2 1831.47  4785.2 1829.49
  4852.0 1827.28  4948.1 1825.44  4956.1 1824.88  4969.5 1823.06  4975.9 1821.67
  4976.4 1821.17  4984.0 1821.17  4984.5 1821.67  4986.4 1822.82  5015.7 1822.94
  5043.9 1826.00  5072.2 1826.48  5142.9 1826.38  5227.8 1827.47  5383.3 1831.94
  5439.9 1834.84  5482.3 1837.65  5510.6 1840.04  5538.9 1844.36  5567.2 1846.87
#Mann=3,-1,0
  4574.3    0.05       0  4975.9    0.05       0  4984.5    0.05       0
Bank Sta=4975.9,4984.5
Exp/Cntr=0.3,0.1

Type RM Length L Ch R = 1,4558,447,447,447
BEGIN DESCRIPTION:
Deadman 59 9.0
END DESCRIPTION:
XS GIS Cut Line= 3
      1635555.00      6856388.00      1636105.00      6856338.00
      1636505.03      6855937.97
#Sta/Elev= 30
  4447.2 1839.43  4507.4 1837.09  4537.6 1836.46  4587.8 1834.00  4617.9 1833.17
  4638.0 1831.82  4648.0 1830.60  4678.1 1830.63  4698.2 1829.56  4828.8 1825.43
  4868.9 1822.30  4909.1 1822.98  4929.2 1822.71  4969.3 1820.57  4975.0 1819.76
  4975.5 1819.26  4983.2 1819.26  4983.7 1819.76  5003.0 1820.72  5013.6 1823.18
  5041.9 1824.76  5098.5 1825.71  5310.6 1827.42  5353.0 1828.45  5395.4 1832.82
  5466.2 1837.68  5494.4 1840.28  5522.7 1844.14  5561.6 1848.18  5565.2 1848.18
#Mann=3,-1,0
  4447.2    0.05       0  4975.0    0.05       0  4983.7    0.05       0
Bank Sta=4975,4983.7
Exp/Cntr=0.3,0.1

Type RM Length L Ch R = 1,4111,231,231,231
BEGIN DESCRIPTION:
Deadman 59 8.0
END DESCRIPTION:
XS GIS Cut Line= 3
      1635554.97      6856587.99      1636205.00      6856738.00
      1636781.59      6856691.12
#Sta/Elev= 30
  4327.5 1839.05  4409.6 1836.05  4419.9 1836.24  4532.8 1831.59  4594.4 1829.61
  4625.1 1827.63  4645.7 1828.23  4676.5 1826.82  4768.8 1824.10  4892.0 1821.61
  4953.6 1821.20  4970.7 1818.80  4975.8 1819.11  4979.9 1818.51  4980.4 1818.01
  4988.3 1818.01  4988.8 1818.51  5074.9 1820.02  5125.0 1822.68  5165.2 1822.11
  5205.3 1824.27  5265.5 1825.69  5315.7 1827.60  5335.7 1829.08  5355.8 1831.34
  5476.2 1840.72  5506.3 1844.19  5545.6 1846.76  5550.7 1846.32  5573.1 1848.15
#Mann=3,-1,0
  4327.5    0.05       0  4979.9    0.05       0  4988.8    0.05       0
Bank Sta=4979.9,4988.8
Exp/Cntr=0.3,0.1

Type RM Length L Ch R = 1,3880,333,333,333
BEGIN DESCRIPTION:
Mapping XS 4c69076b
END DESCRIPTION:
XS GIS Cut Line= 3
      1635685.42      6856733.72      1635966.71      6856910.83
      1636647.31      6856955.97
#Sta/Elev= 30
  4328.9 1833.16  4382.7 1831.05  4440.4 1829.70  4446.6 1828.79  4492.2 1826.87
  4519.3 1825.05  4534.6 1823.30  4549.9 1824.49  4571.1 1823.36  4657.3 1821.24
  4779.9 1821.67  4830.0 1819.96  4920.2 1820.13  4990.3 1818.45  4995.8 1817.18
  5000.8 1817.19  5005.9 1815.65  5006.4 1815.15  5014.3 1815.15  5014.8 1815.65
  5020.4 1815.72  5040.4 1820.64  5120.6 1823.93  5151.5 1825.86  5190.8 1831.09
  5240.9 1835.48  5281.0 1840.29  5291.0 1841.57  5302.2 1843.95  5343.4 1847.01
#Mann=3,-1,0
  4328.9    0.05       0  5005.9    0.05       0  5014.8    0.05       0
Bank Sta=5005.9,5014.8
Exp/Cntr=0.3,0.1

Type RM Length L Ch R = 1,3547,361,361,361
BEGIN DESCRIPTION:
Deadman 59 7.0
END DESCRIPTION:
XS GIS Cut Line= 3
      1635504.96      6856637.97      1636147.26      6857146.94
      1636454.96      6857237.99
#Sta/Elev= 30
  4197.8 1840.20  4368.5 1835.27  4496.7 1830.74  4560.8 1827.78  4589.7 1825.15
  4631.7 1823.54  4645.7 1822.07  4668.2 1822.51  4695.4 1821.15  4759.5 1820.20
  4945.4 1820.50  4959.8 1820.18  4966.2 1819.10  4976.2 1815.84  4976.7 1815.34
  4985.1 1815.84  4988.7 1816.54  5014.1 1817.29  5056.7 1817.06  5088.0 1818.87
  5150.5 1819.70  5183.3 1821.18  5216.6 1824.00  5223.5 1825.88  5244.4 1826.55
  5288.3 1831.15  5321.6 1835.85  5327.8 1839.92  5335.6 1842.33  5338.2 1842.33
#Mann=3,-1,0
  4197.8    0.05       0  4976.2    0.05       0  4985.1    0.05       0
Bank Sta=4976.2,4985.1
Exp/Cntr=0.3,0.1

Type RM Length L Ch R = 1,3186,167,167,167
BEGIN DESCRIPTION:
Deadman 59 6.0
END DESCRIPTION:
XS GIS Cut Line= 3
      1635555.01      6856938.01      1636105.00      6857438.00
      1636455.00      6857338.00
#Sta/Elev= 30
  4256.9 1835.00  4419.4 1827.85  4504.5 1821.58  4540.4 1820.09  4596.4 1818.87
  4702.9 1818.97  4738.3 1818.05  4858.6 1819.24  4929.6 1818.90  4993.1 1817.60
  4996.8 1815.78  5002.8 1815.78  5012.6 1812.95  5013.1 1812.45  5021.6 1812.95
  5031.4 1815.14  5073.0 1814.93  5083.4 1816.75  5089.9 1818.93  5095.1 1818.35
  5104.2 1820.24  5114.6 1821.12  5240.7 1828.20  5260.2 1830.34  5291.4 1832.25
  5308.3 1834.64  5313.5 1834.46  5322.6 1836.48  5342.1 1843.75  5364.2 1844.09
#Mann=3,-1,0
  4256.9    0.05       0  5012.6    0.05       0  5021.6    0.05       0
Bank Sta=5012.6,5021.6
Exp/Cntr=0.3,0.1

Type RM Length L Ch R = 1,3019,316,316,316
BEGIN DESCRIPTION:
Mapping XS ce539615
END DESCRIPTION:
XS GIS Cut Line= 3
      1635636.84      6857164.30      1635938.93      6857570.55
      1636441.23      6857674.48
#Sta/Elev= 30
  4323.8 1825.44  4396.5 1819.82  4475.8 1817.00  4575.9 1816.91  4632.2 1817.71
  4717.7 1817.58  4761.6 1816.98  4886.9 1817.32  4942.2 1816.56  4958.8 1815.85
  4969.0 1815.24  4979.2 1812.58  4995.1 1811.04  4995.6 1810.54  5003.6 1810.54
  5004.1 1811.04  5009.9 1813.66  5037.5 1819.83  5042.6 1819.67  5050.7 1820.72
  5060.9 1820.77  5101.8 1822.79  5163.0 1827.02  5224.3 1829.55  5233.2 1830.36
  5238.3 1830.03  5283.4 1832.69  5288.5 1832.43  5306.0 1833.78  5343.0 1835.31
#Mann=3,-1,0
  4323.8    0.05       0  4995.1    0.05       0  5004.1    0.05       0
Bank Sta=4995.1,5004.1
Exp/Cntr=0.3,0.1

Type RM Length L Ch R = 1,2703,290,290,290
BEGIN DESCRIPTION:
Deadman 59 5.0
END DESCRIPTION:
XS GIS Cut Line= 3
      1635505.00      6857038.01      1635955.00      6857838.00
      1636254.99      6857888.00
#Sta/Elev= 30
  4083.0 1833.82  4134.3 1830.33  4186.3 1829.11  4221.0 1827.20  4333.8 1819.94
  4427.2 1816.59  4501.5 1815.97  4544.8 1816.76  4663.4 1815.84  4831.0 1816.17
  4897.6 1814.14  4920.6 1815.38  4943.5 1815.52  4965.5 1814.07  4971.2 1814.36
  4987.2 1812.91  4992.9 1813.20  4998.0 1811.76  5021.1 1811.03  5028.7 1810.21
  5029.3 1809.59  5029.8 1809.09  5038.3 1809.59  5051.6 1811.73  5061.7 1815.10
  5089.6 1816.09  5094.6 1819.85  5112.4 1819.16  5122.5 1821.35  5305.0 1827.74
#Mann=3,-1,0
  4083.0    0.05       0  5029.3    0.05       0  5038.3    0.05       0
Bank Sta=5029.3,5038.3
Exp/Cntr=0.3,0.1

Type RM Length L Ch R = 1,2413,349,349,349
BEGIN DESCRIPTION:
Mapping XS 655c584d
END DESCRIPTION:
XS GIS Cut Line= 3
      1635404.23      6857452.53      1635669.71      6857867.40
      1636210.94      6858034.23
#Sta/Elev= 30
  4503.0 1817.10  4638.9 1819.68  4696.4 1817.67  4723.5 1815.29  4769.1 1813.49
  4775.0 1814.10  4790.2 1813.27  4796.2 1813.99  4805.5 1813.22  4832.5 1814.15
  4841.8 1813.46  4868.9 1813.63  4877.5 1812.30  4884.1 1813.09  4890.1 1812.61
  4899.3 1814.66  4926.4 1814.19  4941.6 1813.39  4956.8 1810.81  4958.3 1809.58
  4958.8 1809.08  4967.3 1809.58  4978.0 1809.75  4984.4 1811.55  5042.9 1812.43
  5063.9 1813.64  5081.0 1813.18  5113.7 1814.93  5456.1 1822.21  5561.9 1826.95
#Mann=3,-1,0
  4503.0    0.05       0  4958.3    0.03       0  4967.3    0.05       0
Bank Sta=4958.3,4967.3
Exp/Cntr=0.3,0.1

Type RM Length L Ch R = 1,2064,165,165,165
BEGIN DESCRIPTION:
Mapping XS b5021685
END DESCRIPTION:
XS GIS Cut Line= 3
      1635234.04      6857886.50      1635400.74      6858025.41
      1636018.83      6858084.44
#Sta/Elev= 30
  4779.0 1821.97  4788.0 1821.15  4794.5 1821.44  4816.6 1819.51  4837.4 1819.04
  4858.4 1820.03  4866.1 1819.89  4872.6 1820.65  4894.7 1819.89  4929.8 1819.96
  4950.7 1819.02  4958.5 1817.67  4965.0 1817.88  4972.8 1816.84  4979.3 1816.95
  4993.6 1813.63  4996.0 1812.07  5000.6 1812.07  5015.3 1806.49  5015.8 1805.99
  5025.0 1805.99  5025.5 1806.49  5030.4 1807.76  5040.5 1808.39  5080.7 1808.77
  5130.9 1813.08  5178.5 1813.78  5341.8 1814.03  5394.2 1814.58  5616.9 1818.88
#Mann=3,-1,0
  4779.0    0.05       0  5015.3    0.03       0  5025.5    0.05       0
Bank Sta=5015.3,5025.5
Exp/Cntr=0.3,0.1

Type RM Length L Ch R = 1,1899,130,130,130
BEGIN DESCRIPTION:
Mapping XS f50a877a
END DESCRIPTION:
XS GIS Cut Line= 2
      1635265.31      6858195.55      1636147.24      6858101.81
#Sta/Elev= 30
  4810.5 1838.88  4840.4 1838.15  4880.6 1834.33  4910.8 1830.50  4940.9 1824.02
  4951.0 1822.71  4961.0 1820.77  4971.1 1816.77  4991.2 1805.20  4996.2 1803.91
  4996.7 1803.41  5005.9 1803.41  5006.4 1803.91  5020.1 1804.05  5025.1 1805.76
  5031.4 1808.97  5041.5 1810.99  5051.5 1812.05  5061.6 1812.37  5122.7 1812.07
  5192.3 1812.90  5242.6 1812.69  5272.8 1813.49  5292.9 1813.27  5353.2 1813.86
  5584.5 1818.91  5644.9 1820.72  5675.0 1822.07  5683.1 1822.99  5697.4 1823.37
#Mann=3,-1,0
  4810.5    0.05       0  4996.2    0.05       0  5006.4    0.05       0
Bank Sta=4996.2,5006.4
Exp/Cntr=0.3,0.1

Type RM Length L Ch R = 1,1769,415,415,415
BEGIN DESCRIPTION:
Deadman 59 4.0
END DESCRIPTION:
XS GIS Cut Line= 3
      1635405.04      6858337.98      1635505.00      6858288.00
      1636305.00      6858138.00
#Sta/Elev= 30
  4893.9 1836.26  4896.6 1836.26  4902.2 1834.73  4907.8 1834.54  4947.0 1824.80
  4952.5 1823.94  4969.3 1813.67  4974.9 1811.69  4986.6 1804.62  4987.1 1804.12
  4996.3 1804.12  4996.8 1804.62  4997.3 1805.08  5008.2 1805.22  5015.8 1805.92
  5026.0 1807.55  5031.9 1810.13  5037.0 1810.83  5046.4 1811.18  5117.6 1811.06
  5299.9 1812.54  5514.4 1817.02  5605.9 1819.61  5630.5 1820.79  5667.0 1823.66
  5688.2 1824.05  5697.5 1824.92  5740.7 1826.52  5768.7 1828.29  5819.6 1830.29
#Mann=3,-1,0
  4893.9    0.05       0  4986.6    0.05       0  4996.8    0.05       0
Bank Sta=4986.6,4996.8
Exp/Cntr=0.3,0.1

Type RM Length L Ch R = 1,1354,427,427,427
BEGIN DESCRIPTION:
Deadman 59 3.0
END DESCRIPTION:
XS GIS Cut Line= 3
      1635505.01      6858688.00      1635705.00      6858638.00
      1636104.98      6858238.02
#Sta/Elev= 30
  4799.0 1844.62  4801.6 1844.62  4809.3 1841.73  4829.9 1837.90  4850.5 1832.55
  4858.3 1830.04  4863.4 1829.38  4871.1 1826.69  4891.8 1821.58  4899.5 1818.95
  4904.6 1818.24  4912.4 1815.62  4933.0 1809.78  4963.9 1803.03  4976.9 1801.11
  4977.4 1800.61  4986.6 1800.61  4987.1 1801.11  4994.8 1801.94  5008.7 1801.57
  5019.3 1805.08  5033.4 1809.01  5047.6 1811.57  5075.9 1809.29  5118.3 1809.00
  5132.4 1809.69  5174.9 1809.61  5288.0 1811.19  5542.5 1817.86  5570.8 1819.25
#Mann=3,-1,0
  4799.0    0.05       0  4976.9    0.05       0  4987.1    0.05       0
Bank Sta=4976.9,4987.1
Exp/Cntr=0.3,0.1

Type RM Length L Ch R = 1,927,84,84,84
BEGIN DESCRIPTION:
Deadman 59 2.0
END DESCRIPTION:
XS GIS Cut Line= 3
      1635604.98      6859088.01      1635855.00      6858988.00
      1636655.03      6858187.97
#Sta/Elev= 30
  4734.9 1846.68  4803.6 1835.47  4810.3 1832.53  4827.8 1828.02  4857.4 1822.24
  4864.2 1818.81  4881.7 1813.53  4911.3 1808.04  4928.8 1803.09  4930.4 1801.42
  4930.9 1800.92  4940.7 1801.42  4940.9 1804.95  4950.3 1806.95  4959.8 1807.15
  4965.1 1810.48  4982.6 1811.41  4989.4 1810.45  5018.3 1811.87  5074.9 1811.49
  5103.2 1807.15  5173.9 1806.24  5456.7 1811.96  5654.7 1818.22  5824.4 1830.39
  5909.3 1833.26  5937.6 1838.71  6050.7 1839.39  6093.1 1843.44  6135.6 1845.67
#Mann=3,-1,0
  4734.9    0.05       0  4930.4    0.05       0  4940.7    0.05       0
Bank Sta=4930.4,4940.7
Exp/Cntr=0.3,0.1

Type RM Length L Ch R = 1,843,315,315,315
BEGIN DESCRIPTION:
Mapping XS 3158436d
END DESCRIPTION:
XS GIS Cut Line= 3
      1635612.56      6859143.46      1635876.43      6859067.08
      1636267.70      6858852.40
#Sta/Elev= 30
  4745.5 1847.89  4758.4 1845.80  4783.8 1843.04  4789.7 1840.93  4810.5 1837.65
  4851.0 1827.95  4856.2 1827.32  4862.6 1824.54  4883.4 1819.16  4889.8 1816.67
  4914.6 1811.08  4923.4 1808.47  4945.8 1806.18  4956.2 1802.74  4962.3 1799.78
  4962.8 1799.28  4972.1 1799.28  4972.6 1799.78  5008.3 1803.03  5022.2 1803.23
  5026.5 1805.19  5032.2 1806.16  5048.3 1806.81  5070.1 1806.24  5091.9 1803.67
  5098.4 1804.51  5113.7 1804.05  5129.8 1806.53  5292.3 1807.52  5466.5 1810.44
#Mann=3,-1,0
  4745.5    0.05       0  4962.3    0.05       0  4972.6    0.05       0
Bank Sta=4962.3,4972.6
Exp/Cntr=0.3,0.1

Type RM Length L Ch R = 1,528,343,343,343
BEGIN DESCRIPTION:
Mapping XS 51e3e9e6
END DESCRIPTION:
XS GIS Cut Line= 2
      1635668.10      6859487.22      1636250.76      6859223.63
#Sta/Elev= 30
  4684.0 1854.02  4690.2 1852.87  4735.5 1849.82  4788.1 1842.09  4793.6 1841.97
  4811.2 1837.66  4834.3 1833.96  4839.8 1831.55  4856.2 1827.83  4862.9 1825.37
  4878.2 1822.51  4886.0 1819.61  4891.5 1818.83  4914.6 1812.60  4922.1 1809.83
  4937.7 1806.23  4944.0 1803.33  4955.0 1803.43  4960.8 1800.71  4984.2 1799.60
  4984.7 1799.10  4994.5 1799.60  5042.8 1800.17  5053.2 1802.15  5058.7 1802.26
  5064.7 1805.01  5075.7 1805.42  5119.6 1804.78  5163.5 1805.70  5323.5 1806.01
#Mann=3,-1,0
  4684.0    0.05       0  4984.2    0.05       0  4994.5    0.05       0
Bank Sta=4984.2,4994.5
Exp/Cntr=0.3,0.1

Type RM Length L Ch R = 1,185,0,0,0
BEGIN DESCRIPTION:
Deadman 59 1.0
END DESCRIPTION:
XS GIS Cut Line= 3
      1635747.56      6859707.70      1636049.63      6859676.46
      1636754.98      6858638.04
#Sta/Elev= 30
  4687.4 1851.17  4736.6 1845.92  4755.2 1841.95  4785.4 1833.18  4825.4 1817.23
  4830.4 1817.68  4835.6 1813.87  4875.8 1803.06  4924.3 1798.48  4956.3 1798.87
  4966.3 1798.08  4971.2 1796.22  4971.7 1795.72  4981.5 1796.22  4991.1 1797.11
  4993.5 1800.37  5014.5 1802.49  5131.2 1802.32  5267.3 1804.83  5670.1 1806.98
  5900.7 1810.47  5915.6 1812.85  6059.3 1816.90  6089.2 1822.01  6152.2 1829.47
  6182.1 1831.01  6188.1 1833.36  6218.0 1833.50  6224.0 1834.98  6246.4 1835.80
#Mann=3,-1,0
  4687.4    0.05       0  4971.2    0.03       0  4981.5    0.05       0
Bank Sta=4971.2,4981.5
Exp/Cntr=0.3,0.1
