--- Deadman Creek.prj (project) ---

Proj Title=Deadman Creek Base Level Engineering
Current Plan=p01
Default Exp/Contr=0.3,0.1
English Units
Geom File=g01
Flow File=f01
Plan File=p01
BEGIN DESCRIPTION:
Deadman Creek
END DESCRIPTION:

--- Deadman Creek.p01 (plan) ---

Plan Title=Multiple Run
Short Identifier=Multiple
Geom File=g01
Flow File=f01
Subcritical Flow
K Sum by GR= 0
Std Step Tol= 0.01
Critical Tol= 0.01
Num of Std Step Trials= 20
Max Error Tol= 0.3
Flow Tol Ratio= 0.001
Split Flow NTrial= 30
Split Flow Tol= 0.02
Split Flow Ratio= 0.02
Log Output Level= 0
Friction Slope Method= 1
Unsteady Friction Slope Method= 2
Unsteady Bridges Friction Slope Method= 1
Parabolic Critical Depth
Global Vel Dist=  1 , 1 , 1
Global Log Level= 0
CheckData=True
Encroach Param= -1, 0, 0, 0
BEGIN DESCRIPTION:
Multiple Run
END DESCRIPTION:

--- Deadman Creek.f01 (steady flow) ---

Flow Title=Multiple
Number of Profiles=7
Profile Names=10-year,25-year,50-year,1pct_min,100-year,1pct_plu,500-year
River Rch & RM= Deadman Creek,Reach-1,179702
     205     279     338     204     407     811     597
River Rch & RM= Deadman Creek,Reach-1,179445
     269     372     456     279     557    1112     841
River Rch & RM= Deadman Creek,Reach-1,176259
     355     499     619     382     762    1520    1170
River Rch & RM= Deadman Creek,Reach-1,171284
     397     560     697     432     861    1719    1332
River Rch & RM= Deadman Creek,Reach-1,168982
     600     866    1094     686    1369    2732    2176
River Rch & RM= Deadman Creek,Reach-1,164996
     844    1235    1575     996    1988    3966    3211
River Rch & RM= Deadman Creek,Reach-1,158904
    1223    1816    2339    1494    2980    5946    4904
River Rch & RM= Deadman Creek,Reach-1,152393
    1233    1829    2355    1503    2998    5982    4926
River Rch & RM= Deadman Creek,Reach-1,150079
    1585    2370    3068    1967    3925    7831    6510
River Rch & RM= Deadman Creek,Reach-1,144041
    1699    2542    3291    2110    4210    8400    6983
River Rch & RM= Deadman Creek,Reach-1,139143
    1993    2992    3883    2495    4977    9931    8288
River Rch & RM= Deadman Creek,Reach-1,132945
    2400    3634    4745    3065    6115   12200   10295
River Rch & RM= Deadman Creek,Reach-1,129135
    2451    3709    4838    3122    6230   12430   10471
River Rch & RM= Deadman Creek,Reach-1,120906
    2433    3675    4788    3086    6157   12285   10321
River Rch & RM= Deadman Creek,Reach-1,117485
    2536    3830    4991    3217    6418   12806   10758
River Rch & RM= Deadman Creek,Reach-1,108291
    2759    4172    5441    3509    7002   13971   11752
River Rch & RM= Deadman Creek,Reach-1,100641
    2859    4320    5630    3628    7238   14442   12127
River Rch & RM= Deadman Creek,Reach-1,92732
    2941    4439    5781    3723    7428   14820   12424
River Rch & RM= Deadman Creek,Reach-1,87866
    3145    4735    6158    3959    7900   15763   13168
River Rch & RM= Deadman Creek,Reach-1,81529
    3099    4654    6043    3878    7738   15440   12852
River Rch & RM= Deadman Creek,Reach-1,75641
    3101    4654    6041    3876    7734   15431   12835
River Rch & RM= Deadman Creek,Reach-1,70837
    3457    5199    6758    4341    8661   17281   14406
River Rch & RM= Deadman Creek,Reach-1,66259
    3447    5181    6731    4322    8623   17204   14328
River Rch & RM= Deadman Creek,Reach-1,63491
    3471    5214    6772    4346    8672   17303   14401
River Rch & RM= Deadman Creek,Reach-1,61236
    3626    5449    7079    4545    9068   18093   15063
River Rch & RM= Deadman Creek,Reach-1,53764
    3641    5471    7107    4561    9101   18160   15114
River Rch & RM= Deadman Creek,Reach-1,52383
    3650    5478    7110    4560    9099   18154   15085
River Rch & RM= Deadman Creek,Reach-1,47431
    3649    5472    7099    4551    9080   18116   15037
River Rch & RM= Deadman Creek,Reach-1,43171
    4968    7491    9757    6277   12524   24989   20882
River Rch & RM= Deadman Creek,Reach-1,38086
    4971    7490    9752    6271   12512   24965   20842
River Rch & RM= Deadman Creek,Reach-1,32014
    4981    7503    9767    6279   12529   24999   20863
River Rch & RM= Deadman Creek,Reach-1,27793
    4963    7472    9723    6248   12466   24874   20741
River Rch & RM= Deadman Creek,Reach-1,24556
    6185    9348   12201    7862   15688   31301   26237
River Rch & RM= Deadman Creek,Reach-1,24110
    6183    9339   12185    7849   15661   31248   26171
River Rch & RM= Deadman Creek,Reach-1,20536
    6209    9377   12232    7879   15720   31366   26263
River Rch & RM= Deadman Creek,Reach-1,20110
    6201    9357   12200    7853   15669   31264   26147
River Rch & RM= Deadman Creek,Reach-1,17238
    6261    9451   12325    7936   15834   31593   26434
River Rch & RM= Deadman Creek,Reach-1,12439
    6285    9484   12365    7959   15881   31687   26499
River Rch & RM= Deadman Creek,Reach-1,7062
    6547    9884   12891    8301   16562   33045   27650
Boundary for River Rch & Prof#=Deadman Creek,Reach-1,1
Up Type=0
Dn Type=3
Dn Slope=0.0018
Boundary for River Rch & Prof#=Deadman Creek,Reach-1,2
Up Type=0
Dn Type=3
Dn Slope=0.0018
Boundary for River Rch & Prof#=Deadman Creek,Reach-1,3
Up Type=0
Dn Type=3
Dn Slope=0.0018
Boundary for River Rch & Prof#=Deadman Creek,Reach-1,4
Up Type=0
Dn Type=3
Dn Slope=0.0018
Boundary for River Rch & Prof#=Deadman Creek,Reach-1,5
Up Type=0
Dn Type=3
Dn Slope=0.0018
Boundary for River Rch & Prof#=Deadman Creek,Reach-1,6
Up Type=0
Dn Type=3
Dn Slope=0.0018
Boundary for River Rch & Prof#=Deadman Creek,Reach-1,7
Up Type=0
Dn Type=3
Dn Slope=0.0018

--- Deadman Creek.g01 (geometry) ---

Geom Title=Existing Conditions

River Reach=Deadman Creek,Reach-1
Reach XY= 30
      1645005.00      6832438.00      1642506.92      6834893.98
      1642647.78      6841487.69      1641454.70      6842762.88
      1642653.04      6850532.12      1638249.54      6858590.45
      1633565.01      6863527.38      1629548.95      6864646.16
      1620812.81      6871631.81      1620201.45      6879236.53
      1611998.92      6883846.13      1610955.00      6887038.00
      1615215.47      6896197.83      1616907.47      6895893.45
      1616924.60      6897508.17      1619752.94      6898793.85
      1617105.38      6903172.85      1618799.72      6904585.29
      1618458.61      6907886.50      1622452.75      6911493.93
      1621708.54      6914386.53      1623703.38      6914744.03
      1623946.91      6918794.08      1621762.23      6920087.69
      1625152.94      6924143.85      1623656.21      6927877.49
      1627055.00      6933488.00      1627047.19      6936244.19
      1623506.86      6938343.77      1621955.00      6949438.00

Type RM Length L Ch R = 1,179702,257,257,257
BEGIN DESCRIPTION:
Deadman Creek 246.0
END DESCRIPTION:
XS GIS Cut Line= 3
      1644861.94      6832286.63      1645005.15      6832442.86
      1645278.59      6832778.80
#Sta/Elev= 30
  4791.6 1992.35  4801.9 1992.24  4822.9 1990.41  4830.3 1990.31  4879.6 1984.95
  4915.3 1981.78  4929.1 1979.74  4957.3 1977.73  4964.7 1976.78  4969.4 1975.47
  4969.7 1974.97  4973.3 1974.97  4973.5 1975.47  4985.6 1976.35  4993.0 1976.02
  5077.8 1977.79  5092.2 1977.37  5100.1 1976.50  5113.3 1976.68  5135.3 1979.00
  5170.5 1979.98  5184.9 1981.33  5213.6 1982.54  5234.4 1982.80  5291.9 1986.84
  5327.1 1988.34  5341.4 1989.72  5347.9 1989.47  5391.0 1992.41  5436.7 1994.01
#Mann=3,-1,0
  4791.6    0.05       0  4969.4    0.03       0  4973.5    0.05       0
Bank Sta=4969.4,4973.5
Exp/Cntr=0.3,0.1

Type RM Length L Ch R = 1,179445,247,247,247
BEGIN DESCRIPTION:
Mapping XS 9f69b397
END DESCRIPTION:
XS GIS Cut Line= 3
      1644713.50      6832458.51      1644822.86      6832625.15
      1645108.93      6832903.41
#Sta/Elev= 30
  4803.8 1988.02  4812.4 1987.26  4818.4 1987.20  4833.5 1985.70  4869.7 1983.00
  4905.8 1981.13  4926.9 1978.88  4948.0 1977.31  4970.6 1974.59  4982.1 1973.89
  4982.3 1973.39  4985.9 1973.39  4986.2 1973.89  5027.9 1975.35  5105.6 1977.00
  5119.7 1977.73  5126.9 1978.65  5133.9 1978.42  5155.2 1979.94  5176.3 1980.67
  5204.6 1982.91  5225.9 1985.52  5232.9 1985.88  5247.0 1987.57  5275.3 1990.12
  5282.5 1990.25  5331.9 1993.95  5349.1 1994.89  5395.7 1997.30  5402.2 1997.98
#Mann=4,-1,0
  4803.8    0.05       0  4982.1    0.05       0  4986.2    0.05       0
  5349.1    0.12       0
Bank Sta=4982.1,4986.2
Exp/Cntr=0.3,0.1

Type RM Length L Ch R = 1,179198,408,408,408
BEGIN DESCRIPTION:
Mapping XS 0b207a60
END DESCRIPTION:
XS GIS Cut Line= 3
      1644475.67      6832581.25      1644671.58      6832811.07
      1644967.26      6833022.00
#Sta/Elev= 30
  4690.7 1983.86  4695.2 1983.25  4744.6 1982.26  4758.9 1981.65  4779.7 1981.45
  4787.4 1980.82  4822.5 1980.04  4900.5 1976.52  4949.9 1973.26  4969.8 1972.89
  4970.1 1972.39  4973.7 1972.39  4973.9 1972.89  5008.1 1973.41  5070.8 1973.31
  5094.2 1973.74  5107.4 1975.64  5129.8 1977.06  5150.7 1979.39  5156.9 1979.30
  5180.2 1980.99  5201.1 1983.49  5230.3 1986.06  5279.4 1988.55  5287.1 1989.69
  5298.2 1990.31  5301.9 1990.67  5308.0 1990.50  5322.8 1991.55  5355.9 1992.60
#Mann=4,-1,0
  4690.7    0.05       0  4969.8    0.05       0  4973.9    0.05       0
  5298.2    0.12       0
Bank Sta=4969.8,4973.9
Exp/Cntr=0.3,0.1

Type RM Length L Ch R = 1,178790,406,406,406
BEGIN DESCRIPTION:
Mapping XS fa1fc0e7
END DESCRIPTION:
XS GIS Cut Line= 3
      1644212.00      6832961.77      1644471.91      6833099.26
      1644850.31      6833119.97
#Sta/Elev= 30
  4801.1 1984.76  4806.9 1984.52  4828.9 1982.51  4845.3 1980.41  4861.1 1979.36
  4867.3 1978.61  4883.7 1977.68  4889.3 1977.72  4895.0 1976.74  4911.3 1975.66
  4927.7 1973.28  4940.2 1972.25  4962.9 1971.06  4983.4 1970.43  4983.7 1969.93
  4987.3 1969.93  4987.6 1970.43  5043.3 1971.06  5059.7 1971.59  5099.2 1971.46
  5158.3 1971.89  5228.4 1973.54  5248.5 1974.37  5278.5 1976.51  5318.6 1977.83
  5328.6 1978.63  5368.6 1979.78  5378.6 1980.50  5408.7 1981.63  5474.1 1985.90
#Mann=3,-1,0
  4801.1    0.05       0  4983.4    0.03       0  4987.6    0.05       0
Bank Sta=4983.4,4987.6
Exp/Cntr=0.3,0.1

Type RM Length L Ch R = 1,178384,271,271,271
BEGIN DESCRIPTION:
Mapping XS 03f95a40
END DESCRIPTION:
XS GIS Cut Line= 2
      1643950.14      6833421.36      1644930.73      6833449.59
#Sta/Elev= 30
  4545.0 1996.15  4609.9 1993.77  4619.9 1992.75  4649.9 1991.37  4659.9 1990.39
  4689.9 1988.83  4709.9 1987.44  4780.0 1981.53  4810.0 1978.61  4820.0 1977.06
  4830.0 1976.34  4860.0 1973.03  4890.0 1970.28  4920.0 1968.94  4987.9 1968.34
  4988.2 1967.84  4991.9 1967.84  4992.2 1968.34  5040.1 1968.93  5180.1 1972.90
  5220.1 1975.21  5260.2 1978.71  5280.2 1981.02  5296.1 1982.34  5301.1 1982.18
  5310.2 1982.75  5350.2 1983.82  5440.2 1987.81  5460.2 1988.42  5526.0 1989.46
#Mann=3,-1,0
  4545.0    0.05       0  4987.9    0.05       0  4992.2    0.05       0
Bank Sta=4987.9,4992.2
Exp/Cntr=0.3,0.1

Type RM Length L Ch R = 1,178113,238,238,238
BEGIN DESCRIPTION:
Mapping XS dddc5324
END DESCRIPTION:
XS GIS Cut Line= 3
      1644074.42      6833709.55      1644396.57      6833705.79
      1644897.57      6833711.44
#Sta/Elev= 30
  4669.2 1977.85  4689.8 1976.28  4699.8 1975.99  4709.8 1976.07  4719.8 1976.75
  4769.8 1973.49  4849.8 1969.61  4859.8 1969.81  4879.8 1969.40  4939.8 1967.25
  4979.8 1964.57  4999.8 1964.01  5009.8 1964.37  5027.7 1963.61  5028.0 1963.11
  5031.7 1963.11  5032.0 1963.61  5059.8 1963.91  5069.8 1964.37  5079.8 1964.03
  5119.8 1964.31  5199.8 1967.95  5249.8 1970.81  5269.8 1972.38  5309.8 1976.51
  5349.8 1978.30  5379.8 1981.44  5409.8 1983.97  5469.8 1987.65  5492.4 1988.35
#Mann=3,-1,0
  4669.2    0.05       0  5027.7    0.05       0  5032.0    0.05       0
Bank Sta=5027.7,5032
Exp/Cntr=0.3,0.1

Type RM Length L Ch R = 1,177875,262,262,262
BEGIN DESCRIPTION:
Mapping XS b9e16337
END DESCRIPTION:
XS GIS Cut Line= 3
      1644050.02      6833709.58      1644206.32      6833815.04
      1644551.49      6834094.55
#Sta/Elev= 30
  4653.9 1980.34  4684.0 1976.87  4707.9 1975.98  4728.9 1974.02  4734.9 1972.54
  4743.9 1972.19  4749.9 1971.06  4785.9 1969.06  4844.8 1967.24  4851.1 1965.79
  4865.5 1964.66  4879.4 1962.42  4900.7 1960.84  4943.7 1960.08  4950.3 1960.94
  4964.7 1961.24  5012.1 1959.88  5012.4 1959.38  5016.4 1959.88  5028.6 1959.89
  5043.0 1961.81  5063.8 1966.28  5099.0 1969.18  5106.9 1969.14  5113.4 1970.04
  5121.3 1969.62  5135.7 1971.01  5162.9 1975.73  5206.1 1981.19  5286.6 1987.93
#Mann=3,-1,0
  4653.9    0.05       0  5012.1    0.05       0  5016.4    0.05       0
Bank Sta=5012.1,5016.4
Exp/Cntr=0.3,0.1

Type RM Length L Ch R = 1,177613,481,481,481
BEGIN DESCRIPTION:
Deadman Creek 242.0
END DESCRIPTION:
XS GIS Cut Line= 3
      1644005.01      6833638.03      1644105.00      6834038.00
      1644205.02      6834188.04
#Sta/Elev= 30
  4592.1 1990.12  4594.6 1990.12  4602.4 1987.48  4623.0 1986.60  4643.6 1984.19
  4651.3 1982.19  4684.8 1979.99  4715.8 1976.85  4746.7 1972.18  4787.9 1968.20
  4816.3 1966.24  4898.7 1962.49  4903.9 1963.02  4945.1 1961.22  4979.0 1958.18
  4979.3 1957.68  4983.1 1957.68  4983.3 1958.18  4994.1 1959.08  5001.8 1961.35
  5007.4 1961.35  5011.9 1962.51  5032.9 1963.64  5047.9 1965.47  5126.1 1971.49
  5148.6 1974.94  5171.1 1976.79  5177.1 1977.59  5181.7 1979.15  5184.7 1979.15
#Mann=3,-1,0
  4592.1    0.05       0  4979.0    0.05       0  4983.3    0.05       0
Bank Sta=4979,4983.3
Exp/Cntr=0.3,0.1

Type RM Length L Ch R = 1,177132,445,445,445
BEGIN DESCRIPTION:
Deadman Creek 241.0
END DESCRIPTION:
XS GIS Cut Line= 3
      1643655.00      6833888.03      1643655.00      6834138.00
      1643755.01      6834538.02
#Sta/Elev= 30
  4749.9 1978.55  4759.9 1977.77  4789.9 1973.47  4799.9 1972.55  4819.9 1969.64
  4849.9 1966.11  4939.9 1962.29  4949.9 1961.33  4979.9 1956.13  4987.6 1955.58
  4987.9 1955.08  4991.8 1955.08  4992.1 1955.58  5017.9 1956.36  5023.1 1957.52
  5030.8 1956.31  5059.1 1957.52  5092.6 1957.63  5100.4 1958.41  5105.5 1958.11
  5113.3 1959.08  5141.6 1959.55  5216.3 1962.35  5270.4 1964.72  5278.2 1965.71
  5352.9 1968.56  5389.0 1971.13  5394.1 1971.02  5409.6 1973.29  5412.2 1973.29
#Mann=3,-1,0
  4749.9    0.05       0  4987.6    0.05       0  4992.1    0.05       0
Bank Sta=4987.6,4992.1
Exp/Cntr=0.3,0.1

Type RM Length L Ch R = 1,176687,428,428,428
BEGIN DESCRIPTION:
Deadman Creek 240.0
END DESCRIPTION:
XS GIS Cut Line= 3
      1643205.02      6834088.04      1643305.00      6834338.00
      1643705.00      6834738.00
#Sta/Elev= 30
  4731.4 1978.09  4746.2 1977.25  4752.9 1975.92  4800.0 1969.57  4853.9 1964.24
  4902.3 1961.48  4914.5 1959.96  4925.2 1959.29  4946.8 1954.77  4966.0 1954.16
  4966.4 1953.66  4970.3 1953.66  4970.6 1954.16  4985.8 1954.88  5014.8 1955.05
  5028.9 1955.92  5127.9 1956.36  5156.2 1957.28  5226.9 1961.86  5241.0 1962.41
  5297.6 1966.43  5311.7 1966.96  5325.9 1968.41  5382.5 1971.14  5424.9 1975.05
  5439.0 1975.87  5481.4 1979.44  5538.0 1983.14  5552.2 1984.69  5566.3 1985.25
#Mann=3,-1,0
  4731.4    0.05       0  4966.0    0.05       0  4970.6    0.05       0
Bank Sta=4966,4970.6
Exp/Cntr=0.3,0.1

Type RM Length L Ch R = 1,176259,422,422,422
BEGIN DESCRIPTION:
Deadman Creek 239.0
END DESCRIPTION:
XS GIS Cut Line= 3
      1642955.00      6834138.03      1642955.00      6834538.00
      1643355.02      6834888.01
#Sta/Elev= 30
  4599.9 1978.44  4629.9 1976.63  4709.9 1968.33  4739.9 1966.81  4849.9 1958.31
  4919.9 1955.78  4969.9 1952.51  4979.9 1951.48  4987.6 1949.58  4987.9 1949.08
  4991.9 1949.08  4992.2 1949.58  4997.4 1950.99  5007.0 1951.44  5021.2 1951.71
  5042.1 1950.88  5070.6 1951.30  5092.4 1953.10  5141.8 1953.55  5212.5 1955.75
  5262.3 1959.33  5311.7 1964.04  5382.8 1967.71  5438.8 1972.02  5453.1 1970.54
  5460.7 1971.26  5467.3 1972.78  5495.8 1974.87  5524.3 1978.01  5531.4 1978.08
#Mann=3,-1,0
  4599.9    0.05       0  4987.6    0.05       0  4992.2    0.05       0
Bank Sta=4987.6,4992.2
Exp/Cntr=0.3,0.1

Type RM Length L Ch R = 1,175837,466,466,466
BEGIN DESCRIPTION:
Deadman Creek 238.0
END DESCRIPTION:
XS GIS Cut Line= 3
      1642255.03      6834588.01      1642655.00      6834688.00
      1643055.02      6834938.01
#Sta/Elev= 30
  4587.9 1969.81  4605.9 1967.55  4618.8 1967.05  4647.1 1964.64  4680.6 1963.89
  4693.5 1963.03  4711.6 1960.95  4817.2 1952.77  4853.3 1947.87  4886.8 1948.73
  4899.7 1947.89  4907.4 1948.05  4928.0 1949.86  4969.3 1949.29  4977.0 1949.83
  5003.1 1949.19  5005.1 1947.23  5005.6 1946.73  5010.1 1946.73  5010.5 1947.23
  5013.7 1947.24  5023.2 1948.67  5044.4 1948.84  5086.9 1950.48  5217.7 1953.06
  5233.1 1954.10  5312.1 1957.05  5364.0 1960.06  5385.2 1962.19  5471.9 1965.87
#Mann=3,-1,0
  4587.9    0.05       0  5005.1    0.05       0  5010.5    0.05       0
Bank Sta=5005.1,5010.5
Exp/Cntr=0.3,0.1

Type RM Length L Ch R = 1,175371,483,483,483
BEGIN DESCRIPTION:
Deadman Creek 237.0
END DESCRIPTION:
XS GIS Cut Line= 3
      1642204.99      6835288.01      1642605.00      6835038.00
      1643004.98      6834988.00
#Sta/Elev= 30
  4528.5 1970.86  4531.5 1970.86  4536.2 1969.54  4542.1 1969.43  4563.9 1966.56
  4594.0 1963.67  4615.2 1962.95  4630.5 1961.45  4636.4 1961.56  4709.5 1956.56
  4724.9 1953.77  4761.4 1951.23  4803.9 1949.72  4855.8 1946.25  4898.2 1946.55
  4956.0 1945.33  4974.5 1943.02  4975.0 1942.52  4979.5 1942.52  4979.9 1943.02
  4992.5 1944.63  5038.0 1944.81  5050.6 1946.00  5060.7 1947.75  5101.0 1950.17
  5191.7 1954.25  5284.9 1957.46  5332.8 1960.68  5365.5 1961.84  5403.3 1964.61
#Mann=3,-1,0
  4528.5    0.05       0  4974.5    0.05       0  4979.9    0.05       0
Bank Sta=4974.5,4979.9
Exp/Cntr=0.3,0.1

Type RM Length L Ch R = 1,174888,438,438,438
BEGIN DESCRIPTION:
Deadman Creek 236.0
END DESCRIPTION:
XS GIS Cut Line= 3
      1642454.98      6835538.01      1642605.00      6835488.00
      1643221.86      6835309.15
#Sta/Elev= 30
  4836.9 1955.17  4889.6 1950.90  4931.8 1949.27  4942.3 1948.49  4952.9 1945.97
  4974.0 1942.56  4984.5 1941.89  4989.7 1940.16  4990.1 1939.66  4994.7 1939.66
  4995.1 1940.16  4997.6 1940.16  5011.8 1942.18  5017.0 1942.53  5026.3 1942.63
  5067.9 1944.93  5117.7 1944.67  5140.8 1945.24  5161.7 1944.99  5328.2 1950.01
  5349.0 1951.27  5368.4 1951.50  5407.2 1953.30  5412.4 1953.88  5474.0 1956.01
  5494.8 1957.41  5551.9 1959.50  5557.3 1960.34  5578.1 1960.65  5637.3 1964.73
#Mann=3,-1,0
  4836.9    0.05       0  4989.7    0.05       0  4995.1    0.05       0
Bank Sta=4989.7,4995.1
Exp/Cntr=0.3,0.1

Type RM Length L Ch R = 1,174450,434,434,434
BEGIN DESCRIPTION:
Deadman Creek 235.0
END DESCRIPTION:
XS GIS Cut Line= 3
      1642105.04      6835887.99      1642855.00      6835788.00
      1643241.32      6835619.15
#Sta/Elev= 30
  4248.5 1974.00  4285.0 1972.85  4349.3 1967.29  4363.2 1966.94  4490.6 1959.77
  4587.7 1953.30  4692.4 1949.56  4732.7 1947.40  4783.2 1943.47  4803.3 1942.67
  4817.2 1943.30  4873.9 1941.71  4895.4 1941.86  4934.5 1940.09  4963.5 1940.80
  4982.2 1939.42  4982.6 1938.92  4987.2 1938.92  4987.7 1939.42  4995.0 1941.57
  5002.6 1942.90  5136.1 1943.44  5165.4 1944.92  5194.2 1945.56  5241.0 1948.66
  5299.8 1951.46  5368.9 1953.68  5376.2 1954.46  5392.3 1954.62  5426.7 1956.39
#Mann=3,-1,0
  4248.5    0.05       0  4982.2    0.05       0  4987.7    0.05       0
Bank Sta=4982.2,4987.7
Exp/Cntr=0.3,0.1

Type RM Length L Ch R = 1,174016,475,475,475
BEGIN DESCRIPTION:
Deadman Creek 234.0
END DESCRIPTION:
XS GIS Cut Line= 3
      1642305.04      6835988.01      1642705.00      6836088.00
      1643505.03      6836088.00
#Sta/Elev= 30
  4583.1 1961.23  4724.8 1951.12  4771.2 1949.25  4871.7 1943.74  4923.2 1941.97
  4943.8 1940.47  4954.1 1938.63  4969.4 1937.28  4969.8 1936.78  4974.5 1936.78
  4975.0 1937.28  4992.8 1939.00  5075.4 1939.59  5095.4 1939.53  5125.4 1937.85
  5145.4 1938.02  5185.4 1940.15  5205.4 1940.23  5235.4 1938.89  5325.4 1942.78
  5375.4 1947.10  5455.4 1952.60  5495.4 1957.30  5565.4 1962.51  5625.4 1967.67
  5665.4 1971.50  5685.4 1974.73  5705.4 1976.68  5785.4 1980.16  5795.4 1981.16
#Mann=3,-1,0
  4583.1    0.05       0  4969.4    0.03       0  4975.0    0.05       0
Bank Sta=4969.4,4975
Exp/Cntr=0.3,0.1

Type RM Length L Ch R = 1,173541,473,473,473
BEGIN DESCRIPTION:
Deadman Creek 233.0
END DESCRIPTION:
XS GIS Cut Line= 3
      1642155.04      6836138.02      1642855.00      6836388.00
      1643255.03      6836287.99
#Sta/Elev= 30
  4256.1 1971.10  4302.2 1967.08  4309.1 1965.38  4341.0 1961.61  4383.5 1958.00
  4394.6 1956.26  4445.6 1952.89  4481.7 1947.54  4599.6 1940.32  4723.3 1937.69
  4896.9 1938.56  4989.3 1937.33  5001.9 1937.78  5017.4 1935.53  5022.6 1935.90
  5027.5 1935.13  5027.9 1934.63  5033.1 1935.13  5081.8 1936.89  5092.1 1936.61
  5099.9 1937.68  5105.0 1937.50  5112.7 1939.08  5141.1 1942.09  5233.5 1948.77
  5257.1 1949.53  5274.8 1951.06  5352.4 1958.23  5401.1 1961.53  5411.7 1962.25
#Mann=6,-1,0
  4256.1    0.05       0  5027.5    0.05       0  5033.1    0.05       0
  5233.5    0.12       0  5274.8    0.05       0  5401.1    0.12       0
Bank Sta=5027.5,5033.1
Exp/Cntr=0.3,0.1

Type RM Length L Ch R = 1,173068,413,413,413
BEGIN DESCRIPTION:
Deadman Creek 232.0
END DESCRIPTION:
XS GIS Cut Line= 3
      1642105.01      6836238.01      1642455.00      6836588.00
      1642805.03      6836688.01
#Sta/Elev= 30
  4505.9 1969.36  4534.2 1967.41  4576.6 1961.11  4590.7 1959.37  4647.3 1953.59
  4675.6 1951.43  4760.4 1940.55  4802.9 1936.52  4831.2 1935.10  4901.9 1934.94
  4930.2 1934.26  4944.3 1930.89  4955.6 1930.44  4956.1 1929.94  4960.8 1929.94
  4961.3 1930.44  4972.6 1931.81  5003.5 1932.67  5011.3 1934.25  5017.8 1934.29
  5023.0 1933.65  5042.5 1933.91  5051.6 1933.50  5084.1 1934.49  5168.6 1939.35
  5197.2 1940.60  5208.9 1941.53  5265.8 1943.83  5351.2 1947.94  5364.9 1948.63
#Mann=5,-1,0
  4505.9    0.05       0  4955.6    0.05       0  4961.3    0.05       0
  5265.8    0.12       0  5351.2    0.05       0
Bank Sta=4955.6,4961.3
Exp/Cntr=0.3,0.1

Type RM Length L Ch R = 1,172655,452,452,452
BEGIN DESCRIPTION:
Deadman Creek 231.0
END DESCRIPTION:
XS GIS Cut Line= 3
      1641905.04      6836938.00      1642305.00      6836888.00
      1643054.96      6836938.00
#Sta/Elev= 30
  4592.4 1961.89  4622.6 1958.36  4630.2 1955.84  4635.2 1955.45  4642.8 1953.80
  4673.0 1949.12  4743.5 1942.14  4791.4 1935.48  4824.2 1932.47  4834.2 1930.83
  4844.3 1930.71  4904.8 1932.29  4965.2 1932.43  5025.5 1930.72  5042.7 1929.41
  5043.2 1928.91  5048.0 1928.91  5048.4 1929.41  5055.6 1932.10  5065.6 1933.42
  5229.5 1939.23  5336.2 1943.12  5423.8 1945.48  5466.5 1946.94  5486.6 1948.19
  5667.0 1954.63  5697.0 1956.58  5707.1 1956.74  5727.1 1958.32  5747.1 1958.92
#Mann=5,-1,0
  4592.4    0.05       0  5042.7    0.05       0  5048.4    0.05       0
  5229.5    0.12       0  5423.8    0.05       0
Bank Sta=5042.7,5048.4
Exp/Cntr=0.3,0.1

Type RM Length L Ch R = 1,172203,449,449,449
BEGIN DESCRIPTION:
Deadman Creek 230.0
END DESCRIPTION:
XS GIS Cut Line= 3
      1641952.51      6837337.93      1642355.00      6837288.00
      1642755.01      6837087.99
#Sta/Elev= 30
  4598.8 1953.69  4602.6 1953.69  4637.7 1950.47  4642.8 1950.55  4661.8 1948.76
  4782.7 1941.26  4792.8 1940.30  4799.6 1938.77  4804.6 1938.56  4833.1 1935.38
  4843.1 1934.92  4880.5 1931.77  4903.6 1930.49  4923.8 1928.65  4943.9 1927.69
  4958.5 1926.16  4959.0 1925.66  4963.8 1925.66  4964.3 1926.16  5007.2 1927.60
  5012.8 1929.04  5107.8 1931.37  5138.5 1932.51  5214.0 1933.88  5258.7 1935.62
  5264.3 1936.26  5272.7 1936.04  5308.3 1937.48  5420.6 1942.27  5451.6 1943.66
#Mann=5,-1,0
  4598.8    0.05       0  4958.5    0.03       0  4964.3    0.05       0
  5308.3    0.12       0  5420.6    0.05       0
Bank Sta=4958.5,4964.3
Exp/Cntr=0.3,0.1

Type RM Length L Ch R = 1,171754,470,470,470
BEGIN DESCRIPTION:
Deadman Creek 229.0
END DESCRIPTION:
XS GIS Cut Line= 3
      1642204.98      6837738.00      1642505.00      6837688.00
      1642904.97      6837288.03
#Sta/Elev= 30
  4695.6 1940.83  4756.5 1938.56  4845.2 1933.67  4857.8 1932.28  4888.2 1930.50
  4906.0 1928.94  4938.9 1927.21  4949.1 1926.23  4959.2 1924.65  4963.9 1923.18
  4964.4 1922.68  4969.3 1922.68  4969.7 1923.18  4979.5 1924.25  5003.3 1924.95
  5013.9 1925.52  5028.0 1926.79  5070.5 1926.20  5098.8 1926.40  5183.6 1928.36
  5226.0 1930.13  5296.7 1932.11  5339.2 1933.98  5367.5 1935.60  5381.6 1936.72
  5424.0 1938.40  5508.9 1942.46  5551.3 1944.93  5561.9 1945.86  5565.4 1945.86
#Mann=3,-1,0
  4695.6    0.05       0  4963.9    0.05       0  4969.7    0.05       0
Bank Sta=4963.9,4969.7
Exp/Cntr=0.3,0.1

Type RM Length L Ch R = 1,171284,348,348,348
BEGIN DESCRIPTION:
Deadman Creek 228.0
END DESCRIPTION:
XS GIS Cut Line= 3
      1642055.00      6837938.00      1642855.00      6837938.00
      1643005.02      6837837.98
#Sta/Elev= 30
  4205.8 1952.01  4208.3 1952.01  4215.8 1950.68  4225.8 1949.64  4255.8 1947.48
  4315.8 1945.07  4435.8 1938.67  4605.8 1932.10  4715.8 1926.54  4765.8 1925.35
  4855.8 1925.36  4905.8 1924.88  4935.8 1923.96  4952.8 1921.09  4953.3 1920.59
  4958.2 1920.59  4958.7 1921.09  4975.8 1921.66  4995.8 1923.39  5003.3 1924.89
  5008.8 1924.89  5013.3 1926.27  5034.3 1928.79  5064.4 1930.24  5121.5 1935.55
  5150.0 1937.25  5163.5 1939.27  5178.6 1940.81  5183.1 1942.14  5186.1 1942.14
#Mann=3,-1,0
  4205.8    0.05       0  4952.8    0.05       0  4958.7    0.05       0
Bank Sta=4952.8,4958.7
Exp/Cntr=0.3,0.1

Type RM Length L Ch R = 1,170936,484,484,484
BEGIN DESCRIPTION:
Mapping XS b93543b9
END DESCRIPTION:
XS GIS Cut Line= 3
      1642290.57      6838049.95      1642778.22      6838131.61
      1643128.18      6838325.25
#Sta/Elev= 30
  4305.5 1939.82  4380.2 1935.70  4562.3 1928.09  4583.8 1926.61  4688.7 1923.90
  4725.7 1921.67  4749.4 1921.74  4786.5 1923.51  4845.9 1922.08  4889.4 1923.47
  4921.5 1923.22  4933.4 1922.66  4943.3 1921.15  4949.0 1921.71  4967.8 1919.22
  4968.3 1918.72  4973.2 1918.72  4973.7 1919.22  4979.1 1919.53  4986.8 1922.44
  4992.5 1921.92  5008.5 1927.53  5030.3 1927.67  5111.6 1935.37  5133.3 1936.50
  5139.1 1937.78  5155.1 1938.69  5171.1 1941.04  5192.9 1942.98  5199.9 1942.93
#Mann=3,-1,0
  4305.5    0.05       0  4967.8    0.05       0  4973.7    0.05       0
Bank Sta=4967.8,4973.7
Exp/Cntr=0.3,0.1

Type RM Length L Ch R = 1,170452,191,191,191
BEGIN DESCRIPTION:
Mapping XS 85bdde2f
END DESCRIPTION:
XS GIS Cut Line= 3
      1642298.84      6838421.27      1642746.78      6838379.60
      1643191.02      6838345.83
#Sta/Elev= 30
  4692.3 1943.74  4782.7 1937.47  4819.0 1934.16  4879.3 1931.36  4886.9 1930.36
  4939.5 1926.70  4989.7 1921.77  4996.1 1919.67  5009.8 1918.10  5016.9 1916.43
  5017.4 1915.93  5022.4 1915.93  5022.9 1916.43  5029.9 1916.47  5050.0 1919.51
  5138.8 1921.76  5227.5 1921.44  5290.8 1922.12  5320.9 1923.10  5358.6 1927.03
  5363.6 1926.83  5431.2 1934.21  5471.3 1937.64  5489.7 1939.99  5494.8 1939.80
  5501.4 1940.96  5531.5 1943.80  5561.6 1945.36  5581.7 1946.78  5587.7 1947.75
#Mann=3,-1,0
  4692.3    0.05       0  5016.9    0.05       0  5022.9    0.05       0
Bank Sta=5016.9,5022.9
Exp/Cntr=0.3,0.1

Type RM Length L Ch R = 1,170261,382,382,382
BEGIN DESCRIPTION:
Deadman Creek 226.0
END DESCRIPTION:
XS GIS Cut Line= 3
      1642241.58      6838621.79      1642663.44      6838567.10
      1643194.73      6838460.32
#Sta/Elev= 30
  4583.1 1945.00  4651.8 1942.09  4805.2 1930.79  4810.2 1931.05  4884.4 1923.98
  4889.5 1924.06  4949.6 1918.36  4958.6 1916.98  4976.8 1915.83  4977.3 1915.33
  4982.3 1915.33  4982.8 1915.83  5027.3 1918.46  5032.4 1917.41  5078.2 1919.33
  5083.3 1918.91  5173.3 1920.63  5254.9 1923.65  5281.7 1925.84  5286.8 1925.63
  5316.1 1928.37  5332.6 1930.79  5337.7 1930.58  5383.5 1935.02  5388.6 1934.98
  5434.3 1939.85  5485.2 1943.71  5536.1 1946.33  5541.2 1947.37  5550.4 1948.13
#Mann=3,-1,0
  4583.1    0.05       0  4976.8    0.03       0  4982.8    0.05       0
Bank Sta=4976.8,4982.8
Exp/Cntr=0.3,0.1

Type RM Length L Ch R = 1,169879,497,497,497
BEGIN DESCRIPTION:
Deadman Creek 225.0
END DESCRIPTION:
XS GIS Cut Line= 3
      1642291.01      6838994.19      1642606.15      6838934.29
      1643046.24      6838895.23
#Sta/Elev= 30
  4676.0 1931.49  4683.8 1932.04  4700.4 1930.54  4736.0 1929.63  4788.2 1923.64
  4793.3 1923.84  4812.4 1921.47  4822.6 1919.49  4840.4 1914.07  4845.5 1914.88
  4853.1 1913.29  4870.5 1913.27  4871.0 1912.77  4876.0 1912.77  4876.5 1913.27
  4904.0 1914.64  4914.2 1914.53  4944.7 1916.93  4965.1 1917.20  4993.7 1914.16
  5025.7 1914.51  5065.9 1913.94  5075.9 1915.24  5096.0 1919.51  5166.3 1920.22
  5226.5 1921.97  5266.7 1923.87  5367.1 1931.38  5397.2 1935.03  5438.6 1938.81
#Mann=3,-1,0
  4676.0    0.05       0  4870.5    0.03       0  4876.5    0.05       0
Bank Sta=4870.5,4876.5
Exp/Cntr=0.3,0.1

Type RM Length L Ch R = 1,169382,400,400,400
BEGIN DESCRIPTION:
Deadman Creek 224.0
END DESCRIPTION:
XS GIS Cut Line= 3
      1642171.28      6839259.82      1642358.83      6839339.58
      1642955.08      6839322.31
#Sta/Elev= 30
  4796.2 1929.18  4852.3 1927.80  4905.0 1925.01  4928.6 1924.23  4957.7 1921.28
  4963.2 1919.23  4986.8 1914.60  4995.2 1912.39  5000.0 1912.39  5006.2 1910.60
  5032.9 1910.32  5033.4 1909.82  5038.9 1909.82  5039.4 1910.32  5056.2 1911.21
  5066.2 1912.17  5086.2 1914.89  5256.3 1915.44  5276.3 1916.07  5346.3 1916.87
  5386.3 1917.86  5406.3 1918.66  5416.3 1919.69  5436.4 1920.32  5456.4 1921.75
  5476.4 1924.00  5496.4 1925.69  5526.4 1927.56  5556.4 1928.72  5596.5 1929.45
#Mann=3,-1,0
  4796.2    0.05       0  5032.9    0.05       0  5039.4    0.05       0
Bank Sta=5032.9,5039.4
Exp/Cntr=0.3,0.1

Type RM Length L Ch R = 1,168982,396,396,396
BEGIN DESCRIPTION:
Deadman Creek 223.0
END DESCRIPTION:
XS GIS Cut Line= 3
      1642074.87      6839608.75      1642270.21      6839715.54
      1643054.99      6840237.99
#Sta/Elev= 30
  4792.6 1921.22  4821.8 1920.57  4843.6 1918.78  4975.1 1913.90  4990.6 1911.98
  4997.9 1908.97  5011.9 1907.01  5012.4 1906.51  5018.4 1907.01  5027.8 1908.45
  5048.9 1909.57  5063.9 1911.40  5178.1 1909.96  5214.2 1910.24  5229.2 1907.08
  5259.3 1908.59  5280.3 1910.67  5309.3 1911.14  5381.4 1909.55  5445.6 1909.46
  5481.7 1910.38  5511.7 1913.10  5589.8 1917.96  5656.0 1923.62  5683.0 1926.74
  5719.1 1929.72  5749.1 1931.04  5791.2 1935.36  5827.3 1938.09  5958.0 1945.48
#Mann=3,-1,0
  4792.6    0.05       0  5011.9    0.03       0  5018.4    0.05       0
#XS Ineff=2,0
       0                 5180.00    0.00 1918.36
Permanent Ineff=
       F       F
Bank Sta=5011.9,5018.4
Exp/Cntr=0.3,0.1

Type RM Length L Ch R = 1,168586,477,477,477
BEGIN DESCRIPTION:
Deadman Creek 222.0
END DESCRIPTION:
XS GIS Cut Line= 3
      1641505.03      6839988.00      1642205.00      6840088.00
      1642771.37      6840074.95
#Sta/Elev= 30
  4293.5 1936.29  4323.8 1933.51  4364.2 1931.95  4404.6 1928.82  4525.8 1924.82
  4616.7 1920.50  4727.8 1914.06  4758.1 1911.73  4768.2 1910.11  4869.3 1910.10
  4940.0 1907.54  4960.2 1907.46  4970.3 1908.59  5020.6 1905.14  5060.6 1907.76
  5110.6 1908.24  5120.6 1907.73  5127.3 1904.53  5127.8 1904.03  5133.5 1904.03
  5134.0 1904.53  5160.6 1907.38  5170.6 1907.14  5190.6 1908.12  5270.6 1908.50
  5310.7 1907.18  5350.7 1907.42  5380.7 1910.67  5420.7 1913.85  5567.1 1922.67
#Mann=3,-1,0
  4293.5    0.05       0  5127.3    0.03       0  5134.0    0.05       0
#XS Ineff=2,0
    0.00 4980.00 1917.50               0
Permanent Ineff=
       F       F
Bank Sta=5127.3,5134
Exp/Cntr=0.3,0.1

Type RM Length L Ch R = 1,168109,449,449,449
BEGIN DESCRIPTION:
Deadman Creek 221.0
END DESCRIPTION:
XS GIS Cut Line= 3
      1641579.97      6840162.99      1642405.00      6840438.00
      1642604.98      6840388.00
#Sta/Elev= 30
  4135.1 1929.70  4161.5 1929.13  4203.7 1926.51  4288.0 1923.94  4330.1 1921.16
  4351.2 1920.34  4393.4 1917.36  4425.0 1916.07  4583.1 1912.41  4699.1 1910.61
  4772.9 1908.56  4825.6 1907.83  4952.1 1904.55  4962.6 1903.36  4983.7 1902.83
  4989.1 1902.18  4989.6 1901.68  4998.8 1901.68  4999.3 1902.18  5007.3 1902.22
  5015.1 1903.23  5022.8 1905.23  5028.0 1904.93  5035.7 1907.24  5064.0 1910.16
  5069.2 1910.11  5128.5 1917.39  5159.4 1919.59  5187.7 1922.97  5210.9 1925.01
#Mann=3,-1,0
  4135.1    0.05       0  4989.1    0.03       0  4999.3    0.05       0
Bank Sta=4989.1,4999.3
Exp/Cntr=0.3,0.1

Type RM Length L Ch R = 1,167660,497,497,497
BEGIN DESCRIPTION:
Deadman Creek 220.0
END DESCRIPTION:
XS GIS Cut Line= 3
      1641798.87      6840801.48      1642194.69      6840817.10
      1643007.20      6840533.24
#Sta/Elev= 30
  4593.8 1920.10  4609.9 1919.00  4660.0 1917.88  4700.0 1915.90  4770.1 1914.43
  4920.2 1909.52  4940.2 1908.43  4960.2 1906.52  4980.2 1904.31  4987.6 1902.81
  4992.7 1902.81  4999.0 1901.21  5004.3 1901.36  5006.2 1900.42  5006.7 1899.92
  5016.1 1899.92  5016.6 1900.42  5035.3 1901.15  5061.1 1903.57  5128.5 1902.81
  5148.9 1903.61  5265.7 1905.73  5297.4 1906.87  5477.5 1915.59  5647.0 1927.61
  5678.8 1929.20  5784.7 1932.69  5816.1 1934.03  5827.1 1935.38  5850.6 1936.18
#Mann=3,-1,0
  4593.8    0.05       0  5006.2    0.03       0  5016.6    0.05       0
Bank Sta=5006.2,5016.6
Exp/Cntr=0.3,0.1

Type RM Length L Ch R = 1,167163,139,139,139
BEGIN DESCRIPTION:
Deadman Creek 219.0
END DESCRIPTION:
XS GIS Cut Line= 3
      1642255.03      6841287.97      1642355.00      6841188.00
      1642891.35      6840701.36
#Sta/Elev= 30
  4858.4 1914.26  4861.9 1914.26  4900.8 1907.52  4929.1 1899.37  4943.2 1896.38
  5065.2 1895.99  5065.7 1895.49  5075.6 1895.99  5120.4 1896.59  5127.2 1898.67
  5134.6 1898.35  5141.4 1899.10  5148.3 1896.66  5162.3 1896.08  5168.6 1896.63
  5183.9 1901.34  5190.7 1902.06  5269.1 1904.47  5275.8 1905.45  5283.3 1907.89
  5304.2 1911.18  5332.6 1914.08  5353.6 1915.34  5396.1 1915.82  5403.6 1912.05
  5410.3 1909.72  5417.8 1908.37  5566.4 1914.73  5644.2 1919.48  5724.0 1925.90
#Mann=3,-1,0
  4858.4    0.05       0  5065.2    0.03       0  5075.6    0.05       0
Bank Sta=5065.2,5075.6
Exp/Cntr=0.3,0.1

Type RM Length L Ch R = 1,167024,119,119,119
BEGIN DESCRIPTION:
Mapping XS 02125809
END DESCRIPTION:
XS GIS Cut Line= 4
      1642175.96      6841351.90      1642425.67      6841275.46
      1642723.83      6841232.13      1643055.09      6840934.00
#Sta/Elev= 30
  4723.5 1924.33  4732.9 1923.89  4789.3 1918.16  4816.6 1915.27  4837.5 1912.42
  4860.0 1908.95  4868.9 1906.26  4879.4 1905.02  4900.3 1901.50  4910.7 1900.43
  4925.6 1896.39  4952.6 1895.96  5221.2 1895.87  5221.7 1895.37  5231.2 1895.37
  5231.7 1895.87  5311.1 1896.03  5360.4 1897.88  5381.7 1899.96  5395.6 1903.16
  5403.0 1904.29  5431.4 1906.23  5452.4 1908.90  5523.4 1911.50  5615.3 1915.67
  5629.5 1916.59  5637.0 1917.66  5678.8 1920.06  5686.3 1921.05  5731.6 1924.46
#Mann=3,-1,0
  4723.5    0.05       0  5221.2    0.03       0  5231.7    0.05       0
Bank Sta=5221.2,5231.7
Exp/Cntr=0.3,0.1

Type RM Length L Ch R = 1,166905,155,155,155
BEGIN DESCRIPTION:
Mapping XS 72ddc36e
END DESCRIPTION:
XS GIS Cut Line= 6
      1642094.43      6841430.90      1642305.90      6841395.23
      1642522.51      6841367.20      1642728.93      6841344.26
      1642838.51      6841262.71      1643150.97      6841001.06
#Sta/Elev= 30
  4584.6 1926.31  4656.2 1924.23  4691.9 1921.29  4717.0 1920.47  4788.0 1914.12
  4814.9 1909.85  5140.7 1911.14  5201.1 1910.74  5225.2 1907.89  5233.1 1910.38
  5241.5 1909.22  5247.7 1910.85  5291.6 1910.98  5327.0 1909.25  5361.5 1909.28
  5370.2 1907.92  5371.6 1905.72  5372.1 1905.22  5382.1 1905.72  5383.3 1907.42
  5391.1 1905.96  5397.6 1907.93  5412.0 1909.65  5440.6 1906.94  5469.2 1909.30
  5611.0 1916.58  5660.5 1920.17  5709.9 1925.31  5767.2 1929.11  5769.3 1930.11
#Mann=3,-1,0
  4584.6    0.05       0  5371.6    0.05       0  5382.1    0.05       0
Bank Sta=5371.6,5382.1
Exp/Cntr=0.3,0.1

Type RM Length L Ch R = 1,166750,462,462,462
BEGIN DESCRIPTION:
Mapping XS f265a20e
END DESCRIPTION:
XS GIS Cut Line= 4
      1642147.88      6841494.62      1642535.25      6841466.58
      1642677.96      6841446.20      1643181.28      6841275.88
#Sta/Elev= 30
  4525.3 1922.92  4547.6 1920.20  4612.7 1916.07  4662.8 1910.88  4687.0 1909.92
  4712.9 1907.17  4813.2 1900.37  5009.6 1898.76  5039.5 1896.35  5040.0 1895.85
  5050.0 1896.35  5063.9 1898.59  5095.3 1897.36  5100.6 1898.21  5132.1 1898.15
  5158.2 1896.56  5163.5 1898.78  5170.8 1896.98  5194.9 1897.27  5213.1 1899.19
  5221.1 1901.51  5226.4 1900.53  5252.5 1905.06  5339.8 1906.86  5446.4 1913.97
  5504.0 1920.28  5540.7 1923.09  5566.9 1926.67  5572.1 1926.30  5589.2 1928.87
#Mann=3,-1,0
  4525.3    0.05       0  5039.5    0.05       0  5050.0    0.05       0
Bank Sta=5039.5,5050
Exp/Cntr=0.3,0.1

Type RM Length L Ch R = 1,166288,441,441,441
BEGIN DESCRIPTION:
Deadman Creek 217.0
END DESCRIPTION:
XS GIS Cut Line= 3
      1642105.04      6841538.03      1642455.00      6841788.00
      1642855.01      6841988.01
#Sta/Elev= 30
  4574.9 1923.80  4674.4 1914.99  4697.7 1911.82  4760.4 1905.99  4896.8 1898.25
  4932.5 1897.34  4955.8 1897.49  4968.1 1895.58  4976.7 1892.76  4986.2 1892.50
  4986.7 1892.00  4996.2 1892.00  4996.7 1892.50  5001.9 1895.42  5007.8 1895.42
  5013.4 1896.19  5041.3 1895.90  5049.7 1896.97  5063.7 1899.75  5125.2 1899.08
  5139.1 1899.42  5161.6 1898.79  5211.1 1897.97  5264.9 1897.74  5287.3 1898.50
  5295.7 1899.47  5318.0 1904.52  5354.4 1911.29  5376.7 1916.05  5452.2 1924.30
#Mann=5,-1,0
  4574.9    0.05       0  4986.2    0.05       0  4996.7    0.05       0
  5161.6    0.12       0  5211.1    0.05       0
Bank Sta=4986.2,4996.7
Exp/Cntr=0.3,0.1

Type RM Length L Ch R = 1,165847,451,451,451
BEGIN DESCRIPTION:
Deadman Creek 216.0
END DESCRIPTION:
XS GIS Cut Line= 3
      1641855.01      6841888.00      1642205.00      6842088.00
      1642554.98      6842287.99
#Sta/Elev= 30
  4597.1 1928.17  4626.6 1924.24  4669.8 1921.57  4700.8 1917.10  4728.8 1914.19
  4735.3 1912.14  4787.9 1904.98  4852.6 1900.88  4903.8 1899.89  4964.9 1898.53
  4970.7 1897.76  4977.2 1894.90  4987.0 1891.91  4987.5 1891.41  4997.1 1891.41
  4997.6 1891.91  5000.2 1892.63  5029.7 1894.05  5051.3 1893.81  5067.2 1895.03
  5110.3 1895.68  5153.5 1894.87  5184.5 1895.55  5255.8 1894.44  5277.3 1895.11
  5293.2 1896.08  5299.7 1897.55  5358.0 1906.11  5380.3 1907.45  5403.3 1907.94
#Mann=4,-1,0
  4597.1    0.05       0  4903.8    0.12       0  4987.0    0.05       0
  4997.6    0.05       0
Bank Sta=4987,4997.6
Exp/Cntr=0.3,0.1

Type RM Length L Ch R = 1,165396,400,400,400
BEGIN DESCRIPTION:
Deadman Creek 215.0
END DESCRIPTION:
XS GIS Cut Line= 3
      1641954.99      6842087.99      1642355.00      6842488.00
      1642505.02      6842387.99
#Sta/Elev= 30
  4433.5 1904.99  4504.2 1899.63  4589.7 1897.82  4615.8 1897.13  4744.6 1896.19
  4772.9 1895.58  4843.6 1895.48  4857.8 1894.73  4928.5 1894.08  4942.6 1893.38
  4970.9 1893.64  4985.1 1891.84  4990.4 1888.76  4990.9 1888.26  5000.5 1888.26
  5001.0 1888.76  5002.2 1888.76  5006.7 1890.30  5012.7 1889.12  5021.7 1892.21
  5027.7 1891.14  5035.3 1893.58  5042.8 1895.01  5048.8 1894.88  5063.8 1896.16
  5078.8 1898.07  5084.8 1897.62  5099.9 1897.97  5135.9 1899.84  5179.5 1904.00
#Mann=5,-1,0
  4433.5    0.05       0  4589.7    0.12       0  4615.8    0.05       0
  4990.4    0.05       0  5001.0    0.05       0
Bank Sta=4990.4,5001
Exp/Cntr=0.3,0.1

Type RM Length L Ch R = 1,164996,551,551,551
BEGIN DESCRIPTION:
Deadman Creek 214.0
END DESCRIPTION:
XS GIS Cut Line= 3
      1641780.68      6842100.17      1642087.91      6842746.74
      1642192.06      6843066.97
#Sta/Elev= 30
  4404.4 1922.23  4445.1 1920.44  4479.5 1916.28  4490.5 1915.91  4501.6 1913.78
  4512.7 1913.09  4524.3 1910.05  4547.0 1906.88  4615.2 1898.89  4637.9 1897.08
  4704.0 1895.31  4788.0 1893.09  4938.8 1892.20  4961.6 1889.94  4967.1 1887.95
  4977.7 1887.06  4982.7 1885.73  4983.2 1885.23  4996.9 1885.73  5007.0 1887.21
  5012.5 1886.63  5029.7 1893.06  5035.3 1892.37  5052.5 1894.58  5080.7 1894.77
  5190.8 1899.05  5342.4 1902.22  5414.4 1902.88  5419.6 1903.77  5457.0 1905.64
#Mann=5,-1,0
  4404.4    0.05       0  4704.0    0.12       0  4788.0    0.05       0
  4982.7    0.05       0  4996.9    0.05       0
Bank Sta=4982.7,4996.9
Exp/Cntr=0.3,0.1

Type RM Length L Ch R = 1,164445,439,439,439
BEGIN DESCRIPTION:
Deadman Creek 213.0
END DESCRIPTION:
XS GIS Cut Line= 3
      1641504.99      6842387.97      1641555.00      6842638.00
      1642088.75      6843089.38
#Sta/Elev= 30
  4745.4 1915.08  4765.8 1913.39  4776.0 1911.31  4796.4 1909.48  4827.0 1904.76
  4888.2 1898.67  4898.4 1896.96  4918.8 1892.03  4942.3 1883.68  4942.8 1883.18
  4956.0 1883.18  4956.5 1883.68  4969.8 1885.09  4980.0 1887.24  4997.8 1889.14
  5028.4 1889.34  5057.0 1890.80  5092.1 1891.24  5157.0 1890.38  5235.0 1893.14
  5333.8 1892.92  5348.1 1893.63  5354.7 1893.18  5411.8 1893.32  5461.3 1893.96
  5639.3 1898.78  5645.9 1898.32  5674.4 1898.93  5681.4 1899.60  5699.4 1899.44
#Mann=3,-1,0
  4745.4    0.05       0  4942.3    0.03       0  4956.5    0.05       0
Bank Sta=4942.3,4956.5
Exp/Cntr=0.3,0.1

Type RM Length L Ch R = 1,164006,466,466,466
BEGIN DESCRIPTION:
Deadman Creek 212.0
END DESCRIPTION:
XS GIS Cut Line= 3
      1641254.96      6843038.00      1641455.00      6843038.00
      1642555.02      6843238.00
#Sta/Elev= 30
  4800.2 1920.31  4830.2 1917.40  4870.2 1910.62  4910.2 1905.46  4930.2 1899.77
  4960.2 1887.60  4970.2 1885.06  4990.5 1882.17  4991.0 1881.67  5004.4 1881.67
  5004.9 1882.17  5020.6 1883.84  5026.9 1885.47  5032.0 1885.29  5080.3 1888.97
  5112.0 1890.00  5406.8 1892.10  5585.9 1897.80  5702.8 1900.72  5793.0 1907.16
  5884.5 1911.90  5915.0 1914.41  5921.4 1915.85  5926.4 1915.66  5974.7 1920.14
  5979.8 1919.89  6006.5 1922.77  6067.5 1927.27  6108.1 1929.42  6118.3 1929.30
#Mann=3,-1,0
  4800.2    0.05       0  4990.5    0.05       0  5004.9    0.05       0
Bank Sta=4990.5,5004.9
Exp/Cntr=0.3,0.1

Type RM Length L Ch R = 1,163540,462,462,462
BEGIN DESCRIPTION:
Deadman Creek 211.0
END DESCRIPTION:
XS GIS Cut Line= 3
      1641304.99      6843538.00      1641505.00      6843488.00
      1642605.00      6843388.00
#Sta/Elev= 30
  4788.4 1921.53  4791.0 1921.53  4806.5 1917.79  4811.6 1917.78  4847.7 1911.94
  4852.8 1911.70  4860.6 1909.62  4870.9 1908.40  4888.9 1903.25  4912.1 1898.95
  4930.1 1894.40  4935.3 1894.31  4971.4 1882.95  5027.5 1881.76  5028.0 1881.26
  5041.4 1881.26  5041.9 1881.76  5064.9 1883.13  5095.0 1886.93  5105.0 1887.40
  5342.3 1888.82  5416.3 1890.10  5585.0 1895.23  5637.2 1897.50  5687.4 1902.59
  5747.7 1907.21  5828.0 1911.28  5998.7 1926.89  6038.9 1929.31  6099.1 1931.37
#Mann=5,-1,0
  4788.4    0.05       0  5027.5    0.05       0  5041.9    0.05       0
  5342.3    0.12       0  5585.0    0.05       0
Bank Sta=5027.5,5041.9
Exp/Cntr=0.3,0.1

Type RM Length L Ch R = 1,163078,624,624,624
BEGIN DESCRIPTION:
Deadman Creek 210.0
END DESCRIPTION:
XS GIS Cut Line= 3
      1641505.00      6843988.00      1641705.00      6843888.00
      1642304.99      6843638.00
#Sta/Elev= 30
  4781.0 1913.62  4783.8 1913.62  4803.4 1909.85  4811.8 1906.93  4825.7 1904.16
  4870.4 1896.47  4892.8 1889.87  4915.2 1885.13  4937.5 1882.04  4975.0 1879.52
  4975.5 1879.02  4989.0 1879.02  4989.5 1879.52  5026.3 1880.59  5037.1 1881.34
  5048.5 1883.12  5072.3 1885.02  5120.0 1884.53  5173.1 1886.03  5297.1 1887.05
  5380.0 1886.62  5394.6 1888.11  5416.3 1889.08  5486.2 1891.32  5492.1 1892.29
  5502.9 1892.40  5528.0 1894.91  5574.3 1900.43  5640.0 1906.56  5654.6 1907.29
#Mann=5,-1,0
  4781.0    0.05       0  4975.0    0.05       0  4989.5    0.05       0
  5528.0    0.12       0  5574.3    0.05       0
Bank Sta=4975,4989.5
Exp/Cntr=0.3,0.1

Type RM Length L Ch R = 1,162454,73,73,73
BEGIN DESCRIPTION:
Mapping XS e244e1e5
END DESCRIPTION:
XS GIS Cut Line= 6
      1641552.35      6844473.78      1641964.66      6844417.36
      1642220.73      6844252.43      1642212.05      6844117.88
      1641995.04      6843892.19      1642524.56      6843683.85
#Sta/Elev= 30
  4529.7 1914.34  4755.7 1902.56  4796.3 1898.37  4829.4 1891.69  4856.1 1894.21
  5016.2 1892.00  5068.8 1893.44  5089.6 1890.77  5140.4 1893.33  5239.0 1894.84
  5259.1 1893.10  5287.3 1895.67  5359.0 1896.02  5389.2 1892.63  5394.0 1896.43
  5514.5 1896.43  5658.4 1895.02  5701.2 1891.17  5731.0 1894.82  5778.0 1884.32
  5778.5 1883.82  5792.5 1884.32  5823.2 1887.58  5870.9 1885.70  5887.7 1885.64
  5898.9 1889.39  5941.4 1892.07  5984.4 1898.81  6025.3 1900.72  6274.1 1919.62
#Mann=9,-1,0
  4529.7    0.05       0  5016.2    0.12       0  5140.4    0.05       0
  5287.3    0.12       0  5514.5    0.05       0  5778.0    0.05       0
  5792.5    0.05       0  5870.9    0.12       0  6025.3    0.05       0
Bank Sta=5778,5792.5
Exp/Cntr=0.3,0.1

Type RM Length L Ch R = 1,162381,237,237,237
BEGIN DESCRIPTION:
Mapping XS 83fb1f9c
END DESCRIPTION:
XS GIS Cut Line= 3
      1641769.35      6844560.59      1642068.82      6844452.08
      1642680.40      6844096.42
#Sta/Elev= 30
  4696.7 1904.26  4755.9 1902.88  4798.4 1897.90  4810.7 1899.28  4841.3 1892.56
  4897.3 1883.41  4953.2 1878.15  5006.6 1875.47  5007.1 1874.97  5021.1 1875.47
  5041.8 1876.55  5058.0 1880.50  5083.7 1881.00  5138.3 1883.26  5228.5 1882.34
  5255.8 1887.80  5265.3 1886.76  5271.5 1884.75  5287.3 1883.65  5346.0 1883.93
  5351.8 1883.37  5357.8 1879.16  5389.1 1886.30  5404.1 1886.74  5426.3 1885.33
  5438.8 1887.46  5533.9 1891.67  5571.1 1894.64  5645.6 1905.22  5722.7 1911.10
#Mann=5,-1,0
  4696.7    0.05       0  5006.6    0.05       0  5021.1    0.05       0
  5041.8    0.12       0  5083.7    0.05       0
Bank Sta=5006.6,5021.1
Exp/Cntr=0.3,0.1

Type RM Length L Ch R = 1,162144,270,270,270
BEGIN DESCRIPTION:
Deadman Creek 208.0
END DESCRIPTION:
XS GIS Cut Line= 3
      1641904.99      6844638.00      1642205.00      6844638.00
      1642804.98      6844038.02
#Sta/Elev= 30
  4705.7 1900.21  4735.7 1896.95  4785.7 1887.12  4815.7 1883.75  4855.7 1881.60
  4875.7 1878.91  4905.7 1877.53  4965.7 1876.98  4985.7 1877.69  4995.9 1876.71
  4996.4 1876.21  5010.5 1876.71  5062.3 1878.69  5090.6 1881.14  5189.6 1883.46
  5203.7 1884.82  5217.8 1888.09  5232.0 1884.56  5288.5 1877.34  5302.7 1877.28
  5331.0 1885.86  5444.1 1887.97  5514.8 1892.32  5557.2 1896.29  5606.7 1902.93
  5670.4 1908.64  5712.8 1910.78  5797.7 1918.97  5825.9 1922.67  5854.2 1924.62
#Mann=3,-1,0
  4705.7    0.05       0  4995.9    0.03       0  5010.5    0.05       0
Bank Sta=4995.9,5010.5
Exp/Cntr=0.3,0.1

Type RM Length L Ch R = 1,161874,303,303,303
BEGIN DESCRIPTION:
Deadman Creek 207.0
END DESCRIPTION:
XS GIS Cut Line= 3
      1641804.96      6844787.99      1642316.22      6844873.09
      1643106.15      6844721.18
#Sta/Elev= 30
  4492.1 1901.32  4623.9 1894.23  4715.2 1884.05  4786.1 1879.84  4836.8 1880.55
  4885.2 1877.55  4968.6 1878.17  5007.0 1875.51  5029.5 1876.68  5064.5 1876.90
  5070.3 1875.76  5090.6 1876.88  5093.5 1875.15  5094.0 1874.65  5108.1 1875.15
  5151.7 1881.31  5173.5 1881.25  5220.3 1883.52  5284.1 1883.02  5324.2 1885.57
  5329.3 1884.58  5406.3 1884.41  5518.3 1895.45  5569.2 1902.67  5640.5 1909.28
  5660.9 1911.94  5697.9 1918.95  5749.8 1925.06  5754.9 1924.66  5814.8 1929.68
#Mann=3,-1,0
  4492.1    0.05       0  5093.5    0.03       0  5108.1    0.05       0
Bank Sta=5093.5,5108.1
Exp/Cntr=0.3,0.1

Type RM Length L Ch R = 1,161571,330,330,330
BEGIN DESCRIPTION:
Mapping XS 0132a72b
END DESCRIPTION:
XS GIS Cut Line= 3
      1641883.03      6845079.87      1642216.35      6845157.99
      1642919.42      6845053.83
#Sta/Elev= 30
  4415.0 1888.43  4458.1 1886.42  4520.6 1881.81  4571.1 1879.80  4632.7 1878.84
  4806.5 1879.36  4897.5 1878.14  4958.2 1875.85  4968.3 1873.78  4981.1 1872.97
  4981.6 1872.47  4995.8 1872.97  5008.7 1874.14  5028.9 1873.16  5051.4 1875.52
  5079.5 1877.88  5109.8 1881.55  5150.2 1884.18  5235.9 1886.73  5291.8 1889.06
  5332.2 1893.10  5337.3 1894.32  5342.3 1894.09  5392.9 1901.37  5401.7 1903.25
  5406.8 1902.96  5413.1 1904.41  5433.3 1906.89  5463.4 1913.32  5468.1 1913.32
#Mann=5,-1,0
  4415.0    0.05       0  4981.1    0.05       0  4995.8    0.05       0
  5051.4    0.12       0  5235.9    0.05       0
Bank Sta=4981.1,4995.8
Exp/Cntr=0.3,0.1

Type RM Length L Ch R = 1,161241,330,330,330
BEGIN DESCRIPTION:
Deadman Creek 206.0
END DESCRIPTION:
XS GIS Cut Line= 3
      1641791.06      6845159.55      1642505.00      6845438.00
      1642804.98      6845438.00
#Sta/Elev= 30
  4233.8 1887.98  4273.2 1885.87  4322.2 1884.27  4334.6 1883.13  4442.0 1879.43
  4645.9 1877.90  4708.0 1878.32  4828.4 1876.75  4846.6 1877.37  4852.0 1876.33
  4876.5 1876.70  4906.3 1875.86  4925.0 1874.40  4946.5 1874.26  4967.9 1873.36
  4990.6 1873.40  4997.4 1871.60  5002.6 1871.60  5012.8 1869.87  5013.3 1869.37
  5027.0 1869.37  5027.5 1869.87  5030.1 1871.77  5040.1 1874.94  5060.1 1878.95
  5190.1 1891.21  5230.1 1898.67  5290.1 1908.14  5297.6 1910.02  5300.1 1910.02
#Mann=3,-1,0
  4233.8    0.05       0  5012.8    0.05       0  5027.5    0.05       0
Bank Sta=5012.8,5027.5
Exp/Cntr=0.3,0.1

Type RM Length L Ch R = 1,160911,367,367,367
BEGIN DESCRIPTION:
Mapping XS 3471034c
END DESCRIPTION:
XS GIS Cut Line= 4
      1641665.15      6845207.27      1642220.73      6845606.60
      1642455.11      6845771.53      1642837.09      6845767.19
#Sta/Elev= 30
  4124.5 1890.01  4268.7 1884.23  4310.4 1882.98  4354.6 1882.56  4360.8 1881.79
  4390.2 1880.55  4461.4 1879.12  4555.3 1878.84  4641.5 1877.44  4734.0 1877.83
  4899.5 1874.98  4941.9 1873.30  4948.4 1872.35  4955.4 1868.68  4955.9 1868.18
  4969.7 1868.18  4970.2 1868.68  4971.5 1870.97  4985.1 1870.35  4992.4 1871.17
  4998.5 1871.02  5034.2 1872.27  5063.8 1875.58  5084.8 1878.80  5097.7 1879.33
  5105.2 1880.22  5275.2 1887.93  5315.2 1892.90  5415.2 1894.24  5477.3 1896.54
#Mann=3,-1,0
  4124.5    0.05       0  4955.4    0.05       0  4970.2    0.05       0
Bank Sta=4955.4,4970.2
Exp/Cntr=0.3,0.1
