HEC-RAS study Deadman Creek.prj: Deadman Creek Base Level Engineering

--- Deadman Creek.g01 (geometry) --- (continued)

Type RM Length L Ch R = 1,160544,706,706,706
BEGIN DESCRIPTION:
Mapping XS bbfb9208
END DESCRIPTION:
XS GIS Cut Line= 3
      1641500.23      6845571.87      1642246.78      6846057.99
      1642989.00      6846062.33
#Sta/Elev= 30
  4226.1 1887.69  4341.6 1882.05  4589.3 1874.33  4637.5 1874.39  4661.4 1873.24
  4697.2 1875.34  4733.0 1874.86  4776.4 1875.82  4804.6 1875.46  4869.9 1872.98
  4921.3 1873.46  4948.3 1867.78  4956.0 1867.23  4956.5 1866.73  4970.8 1867.23
  4978.6 1869.18  4993.7 1870.71  5029.9 1871.77  5066.2 1871.43  5079.0 1872.38
  5117.0 1872.87  5135.2 1874.79  5155.2 1875.74  5405.2 1880.12  5575.2 1884.11
  5595.2 1885.12  5615.2 1887.34  5685.2 1890.75  5785.2 1896.94  5859.2 1902.63
#Mann=3,-1,0
  4226.1    0.05       0  4956.0    0.03       0  4970.8    0.05       0
Bank Sta=4956,4970.8
Exp/Cntr=0.3,0.1

Type RM Length L Ch R = 1,159838,378,378,378
BEGIN DESCRIPTION:
Deadman Creek 205.0
END DESCRIPTION:
XS GIS Cut Line= 3
      1641305.01      6846238.00      1641905.00      6846388.00
      1643088.74      6846153.48
#Sta/Elev= 30
  4388.7 1896.91  4512.4 1884.01  4612.9 1877.52  4695.3 1874.71  4700.5 1875.19
  4893.8 1872.77  4914.4 1870.80  4947.9 1869.34  4955.6 1867.90  4989.4 1866.94
  4989.9 1866.44  5004.3 1866.94  5017.3 1868.20  5037.9 1868.21  5058.1 1870.00
  5129.5 1871.65  5211.0 1872.60  5313.0 1872.58  5567.8 1876.35  5639.2 1876.59
  5883.9 1882.25  5934.8 1885.75  5996.0 1888.44  6026.6 1891.31  6057.0 1892.47
  6067.4 1893.82  6097.9 1895.01  6159.1 1899.63  6169.7 1901.20  6213.9 1903.68
#Mann=3,-1,0
  4388.7    0.05       0  4989.4    0.05       0  5004.3    0.05       0
Bank Sta=4989.4,5004.3
Exp/Cntr=0.3,0.1

Type RM Length L Ch R = 1,159460,96,96,96
BEGIN DESCRIPTION:
Deadman Creek 204.0
END DESCRIPTION:
XS GIS Cut Line= 3
      1640820.45      6846757.18      1642046.91      6846721.29
      1642965.12      6846502.95
#Sta/Elev= 30
  3782.6 1923.94  3857.2 1919.49  3928.9 1914.21  4007.2 1907.06  4047.3 1902.56
  4107.3 1898.20  4157.3 1892.84  4237.3 1886.39  4367.4 1878.89  4447.4 1875.32
  4597.5 1872.38  4847.6 1871.30  4897.6 1868.88  4951.8 1867.38  4967.7 1864.65
  4980.2 1863.91  4980.7 1863.41  4995.1 1863.91  5059.0 1869.74  5091.8 1870.90
  5128.8 1871.31  5265.6 1869.75  5295.4 1870.39  5316.0 1871.89  5326.3 1871.48
  5344.8 1872.76  5392.2 1872.23  5434.3 1873.17  5675.7 1874.49  5953.4 1880.20
#Mann=3,-1,0
  3782.6    0.05       0  4980.2    0.05       0  4995.1    0.05       0
Bank Sta=4980.2,4995.1
Exp/Cntr=0.3,0.1

Type RM Length L Ch R = 1,159364,460,460,460
BEGIN DESCRIPTION:
Mapping XS 2f5ce723
END DESCRIPTION:
XS GIS Cut Line= 4
      1640910.27      6846840.94      1641783.68      6846834.96
      1642501.59      6846766.16      1642926.33      6846535.84
#Sta/Elev= 30
  3834.3 1917.78  3859.0 1916.87  3899.0 1914.10  4009.0 1902.36  4059.0 1898.73
  4109.0 1893.72  4159.0 1889.71  4209.0 1886.62  4259.0 1882.51  4339.0 1878.25
  4489.0 1873.42  4609.0 1871.06  4839.7 1870.53  4869.8 1868.33  4910.0 1868.71
  4941.5 1867.59  4972.8 1864.41  4973.3 1863.91  4987.7 1864.41  5000.4 1864.58
  5020.5 1866.25  5030.5 1865.58  5044.2 1867.16  5050.6 1868.78  5080.8 1870.20
  5241.5 1868.91  5357.1 1871.50  5717.2 1873.99  5807.8 1875.36  5912.1 1878.41
#Mann=3,-1,0
  3834.3    0.05       0  4972.8    0.05       0  4987.7    0.05       0
Bank Sta=4972.8,4987.7
Exp/Cntr=0.3,0.1

Type RM Length L Ch R = 1,158904,411,411,411
BEGIN DESCRIPTION:
Deadman Creek 203.0
END DESCRIPTION:
XS GIS Cut Line= 4
      1640979.51      6846951.61      1641819.30      6846911.20
      1642301.17      6847181.95      1642854.96      6847437.98
#Sta/Elev= 30
  3605.3 1915.47  3700.9 1905.09  3785.3 1898.30  3811.0 1894.94  3881.1 1888.91
  4041.3 1879.80  4211.5 1872.91  4381.7 1869.97  4653.6 1870.13  4777.9 1868.51
  4888.5 1866.52  4896.5 1864.42  4911.4 1863.89  4961.6 1864.20  4981.9 1860.11
  4982.4 1859.61  5001.5 1860.11  5036.1 1863.62  5068.2 1864.61  5102.2 1867.55
  5216.8 1870.35  5278.4 1875.58  5344.5 1884.75  5377.3 1886.49  5465.7 1894.52
  5548.9 1899.70  5571.8 1902.32  5594.7 1906.06  5600.2 1908.44  5608.9 1908.97
#Mann=3,-1,0
  3605.3    0.05       0  4981.9    0.05       0  5001.5    0.05       0
Bank Sta=4981.9,5001.5
Exp/Cntr=0.3,0.1

Type RM Length L Ch R = 1,158493,477,477,477
BEGIN DESCRIPTION:
Deadman Creek 202.0
END DESCRIPTION:
XS GIS Cut Line= 3
      1641505.02      6847488.00      1642055.00      6847488.00
      1642655.02      6847488.00
#Sta/Elev= 30
  4450.7 1879.39  4600.7 1873.78  4660.7 1872.19  4760.7 1867.60  4850.7 1865.15
  4880.7 1863.58  4940.7 1864.83  4950.7 1865.61  4970.7 1863.75  4980.7 1860.45
  4990.7 1859.03  5009.7 1857.46  5010.2 1856.96  5027.0 1856.96  5027.5 1857.46
  5040.7 1859.29  5060.7 1863.10  5070.7 1864.05  5100.7 1864.15  5190.7 1868.40
  5280.7 1869.94  5370.7 1870.08  5410.7 1870.76  5430.7 1871.87  5450.7 1871.99
  5460.7 1872.56  5470.7 1874.27  5490.7 1876.27  5530.7 1883.40  5600.7 1889.51
#Mann=3,-1,0
  4450.7    0.05       0  5009.7    0.05       0  5027.5    0.05       0
Bank Sta=5009.7,5027.5
Exp/Cntr=0.3,0.1

Type RM Length L Ch R = 1,158016,468,468,468
BEGIN DESCRIPTION:
Deadman Creek 201.0
END DESCRIPTION:
XS GIS Cut Line= 3
      1641275.90      6847846.19      1641855.00      6847888.00
      1642869.63      6847710.76
#Sta/Elev= 30
  4419.7 1895.15  4514.2 1885.98  4559.2 1882.51  4639.4 1878.55  4819.8 1872.55
  4890.0 1869.03  4910.1 1866.69  4920.1 1863.61  4928.0 1859.98  4933.0 1859.62
  4940.1 1857.49  4952.2 1855.62  4952.6 1855.12  4967.6 1855.12  4968.0 1855.62
  4990.3 1860.73  4997.8 1861.73  5061.2 1863.35  5081.5 1864.28  5087.0 1865.41
  5162.7 1866.54  5193.2 1865.67  5558.6 1868.48  5680.4 1870.93  5726.4 1873.47
  5751.5 1873.42  5792.1 1877.72  5822.6 1880.03  5883.5 1888.22  6030.3 1901.24
#Mann=3,-1,0
  4419.7    0.05       0  4952.2    0.05       0  4968.0    0.05       0
Bank Sta=4952.2,4968
Exp/Cntr=0.3,0.1

Type RM Length L Ch R = 1,157548,482,482,482
BEGIN DESCRIPTION:
Deadman Creek 200.0
END DESCRIPTION:
XS GIS Cut Line= 3
      1641199.54      6848348.31      1641805.00      6848338.00
      1643111.32      6848106.04
#Sta/Elev= 30
  4394.2 1906.21  4559.7 1889.60  4705.3 1879.00  4739.7 1877.79  4849.7 1869.38
  4899.7 1867.41  4919.7 1867.66  4939.7 1865.83  4969.7 1858.03  4979.7 1858.29
  4989.8 1855.62  4990.2 1855.12  5005.7 1855.62  5020.1 1857.41  5026.7 1859.45
  5050.5 1858.97  5070.8 1861.76  5131.8 1860.99  5223.2 1863.08  5661.3 1866.31
  5822.4 1869.00  5984.9 1873.41  6000.4 1874.78  6059.5 1876.37  6113.5 1880.34
  6167.5 1886.15  6177.9 1888.65  6198.2 1891.19  6279.5 1898.22  6326.5 1904.86
#Mann=3,-1,0
  4394.2    0.05       0  4989.8    0.05       0  5005.7    0.05       0
Bank Sta=4989.8,5005.7
Exp/Cntr=0.3,0.1

Type RM Length L Ch R = 1,157066,498,498,498
BEGIN DESCRIPTION:
Deadman Creek 199.0
END DESCRIPTION:
XS GIS Cut Line= 3
      1641305.04      6848887.99      1641905.00      6848788.00
      1643244.56      6848393.07
#Sta/Elev= 30
  4392.3 1910.46  4420.1 1905.73  4486.0 1900.41  4541.8 1892.86  4564.6 1891.31
  4584.9 1888.02  4736.9 1875.97  4785.1 1870.37  4851.0 1864.60  4878.9 1857.94
  4899.2 1856.71  4939.7 1856.76  4960.0 1855.88  4967.6 1854.30  4980.3 1855.86
  4990.4 1855.14  4990.5 1854.25  4990.9 1853.75  5006.3 1854.25  5022.4 1858.01
  5050.5 1860.98  5083.8 1859.99  5209.0 1860.51  5646.9 1863.51  5863.8 1867.52
  6063.9 1873.16  6157.8 1878.00  6241.2 1885.71  6289.7 1892.41  6397.1 1900.98
#Mann=3,-1,0
  4392.3    0.05       0  4990.5    0.05       0  5006.3    0.05       0
Bank Sta=4990.5,5006.3
Exp/Cntr=0.3,0.1

Type RM Length L Ch R = 1,156568,449,449,449
BEGIN DESCRIPTION:
Deadman Creek 198.0
END DESCRIPTION:
XS GIS Cut Line= 3
      1641704.97      6849438.02      1641905.00      6849288.00
      1643515.40      6848497.24
#Sta/Elev= 30
  4740.9 1898.47  4798.2 1887.81  4890.9 1878.62  4940.9 1869.43  4948.2 1867.06
  4954.5 1867.18  4969.1 1864.58  4983.6 1860.16  4987.8 1856.68  4993.7 1856.68
  4999.4 1853.40  5003.3 1848.57  5003.8 1848.07  5023.1 1848.57  5035.5 1852.59
  5080.1 1857.68  5111.8 1858.90  5409.7 1857.99  5826.5 1862.24  6038.1 1866.90
  6171.8 1870.81  6194.1 1872.62  6275.2 1875.76  6382.1 1878.09  6427.1 1882.56
  6539.5 1890.83  6573.1 1895.20  6628.6 1899.78  6695.4 1907.73  6785.0 1920.58
#Mann=3,-1,0
  4740.9    0.05       0  5003.3    0.05       0  5023.1    0.05       0
Bank Sta=5003.3,5023.1
Exp/Cntr=0.3,0.1

Type RM Length L Ch R = 1,156119,480,480,480
BEGIN DESCRIPTION:
Deadman Creek 197.0
END DESCRIPTION:
XS GIS Cut Line= 3
      1641854.97      6849738.01      1642155.00      6849638.00
      1643577.90      6848950.37
#Sta/Elev= 30
  4688.6 1898.72  4751.9 1887.95  4783.5 1883.54  4836.2 1879.00  4899.4 1868.90
  4920.5 1866.44  4952.2 1851.69  4963.3 1845.63  4963.8 1845.13  4983.1 1845.63
  4994.3 1848.27  5002.2 1852.21  5007.6 1852.21  5013.0 1854.87  5032.9 1856.25
  5058.6 1856.17  5086.7 1857.55  5103.8 1856.36  5273.1 1855.58  5837.8 1862.40
  6037.8 1866.46  6226.6 1872.02  6261.4 1873.81  6284.0 1875.94  6368.9 1879.34
  6382.1 1880.85  6436.6 1883.31  6448.7 1884.87  6459.2 1884.61  6585.2 1892.04
#Mann=5,-1,0
  4688.6    0.05       0  4963.3    0.05       0  4983.1    0.05       0
  5013.0    0.12       0  5032.9    0.05       0
Bank Sta=4963.3,4983.1
Exp/Cntr=0.3,0.1

Type RM Length L Ch R = 1,155639,544,544,544
BEGIN DESCRIPTION:
Deadman Creek 196.0
END DESCRIPTION:
XS GIS Cut Line= 3
      1642004.97      6849987.99      1642255.00      6850088.00
      1644020.30      6849966.00
#Sta/Elev= 30
  4725.4 1870.66  4818.3 1864.58  4854.7 1858.06  4877.6 1855.30  4955.6 1854.42
  4962.4 1850.97  4975.4 1847.21  4975.9 1846.71  4995.2 1847.21  5044.8 1853.45
  5084.9 1854.83  5115.0 1854.66  5175.1 1851.89  5185.1 1852.74  5205.2 1851.14
  5211.2 1849.64  5216.2 1851.20  5225.2 1849.87  5275.4 1853.15  5385.6 1852.37
  5435.7 1854.05  5546.0 1854.20  5797.0 1858.95  6117.4 1860.05  6147.4 1862.61
  6230.1 1864.07  6247.7 1861.77  6257.7 1861.76  6367.7 1868.04  6764.2 1884.29
#Mann=3,-1,0
  4725.4    0.05       0  4975.4    0.05       0  4995.2    0.05       0
Bank Sta=4975.4,4995.2
Exp/Cntr=0.3,0.1

Type RM Length L Ch R = 1,155095,572,572,572
BEGIN DESCRIPTION:
Deadman Creek 195.0
END DESCRIPTION:
XS GIS Cut Line= 3
      1641654.99      6850037.99      1642655.00      6850438.00
      1643455.02      6850988.02
#Sta/Elev= 30
  3930.4 1895.50  3969.5 1889.30  4023.3 1884.20  4092.0 1878.52  4106.8 1879.86
  4113.5 1876.80  4124.3 1874.68  4160.6 1873.07  4454.1 1851.12  4566.6 1853.97
  4869.0 1852.78  4914.6 1851.89  4938.8 1848.67  4944.2 1849.13  4953.6 1845.80
  4958.2 1845.79  4958.7 1845.29  4978.6 1845.79  4992.6 1849.34  4998.0 1848.43
  5010.5 1849.99  5014.9 1852.84  5021.0 1850.69  5050.7 1854.94  5071.7 1853.90
  5165.2 1857.34  5474.9 1860.33  5639.3 1863.43  5797.6 1867.94  5978.3 1875.08
#Mann=5,-1,0
  3930.4    0.05       0  4566.6    0.12       0  4869.0    0.05       0
  4958.2    0.05       0  4978.6    0.05       0
Bank Sta=4958.2,4978.6
Exp/Cntr=0.3,0.1

Type RM Length L Ch R = 1,154523,560,560,560
BEGIN DESCRIPTION:
Deadman Creek 194.0
END DESCRIPTION:
XS GIS Cut Line= 3
      1641454.97      6849937.97      1642255.00      6850688.00
      1643355.03      6851788.03
#Sta/Elev= 30
  3903.8 1916.75  4024.2 1905.91  4116.1 1901.73  4215.2 1886.61  4356.4 1878.67
  4370.6 1874.82  4554.7 1862.28  4625.5 1852.68  4731.5 1851.30  4738.8 1848.56
  4753.0 1847.62  4781.1 1851.18  4936.7 1850.72  4958.2 1846.55  4965.0 1842.72
  4969.7 1842.30  4970.1 1841.80  4986.1 1842.30  4986.5 1844.84  5099.4 1852.41
  5707.5 1855.87  5933.8 1859.98  6075.2 1864.75  6131.8 1869.64  6174.2 1876.28
  6287.4 1886.19  6358.1 1899.70  6428.8 1909.23  6513.6 1917.35  6556.1 1917.82
#Mann=3,-1,0
  3903.8    0.05       0  4969.7    0.05       0  4986.1    0.05       0
Bank Sta=4969.7,4986.1
Exp/Cntr=0.3,0.1

Type RM Length L Ch R = 1,153963,570,570,570
BEGIN DESCRIPTION:
Deadman Creek 193.0
END DESCRIPTION:
XS GIS Cut Line= 3
      1641255.04      6850538.03      1641805.00      6850938.00
      1643204.98      6851887.99
#Sta/Elev= 30
  4319.2 1896.95  4355.9 1893.43  4412.3 1884.35  4441.6 1881.34  4518.9 1877.96
  4563.0 1872.64  4891.4 1859.13  4920.8 1856.11  4941.7 1852.37  4956.3 1848.87
  4971.0 1842.70  4980.4 1840.87  4980.8 1840.37  4996.8 1840.87  4999.2 1843.21
  5012.7 1845.22  5057.6 1848.08  5265.1 1847.73  5417.0 1849.88  5863.1 1851.52
  6186.6 1858.70  6267.4 1863.39  6330.3 1874.76  6375.2 1877.53  6432.1 1883.46
  6468.0 1888.16  6510.0 1897.40  6569.8 1907.06  6654.9 1915.27  6691.1 1916.09
#Mann=3,-1,0
  4319.2    0.05       0  4980.4    0.05       0  4996.8    0.05       0
Bank Sta=4980.4,4996.8
Exp/Cntr=0.3,0.1

Type RM Length L Ch R = 1,153393,581,581,581
BEGIN DESCRIPTION:
Deadman Creek 192.0
END DESCRIPTION:
XS GIS Cut Line= 3
      1640855.03      6850688.03      1641605.00      6851438.00
      1643005.04      6852088.02
#Sta/Elev= 30
  3940.4 1909.91  4081.8 1897.83  4180.8 1891.73  4322.2 1877.97  4392.9 1874.05
  4407.0 1874.91  4421.2 1871.74  4845.5 1858.40  4930.3 1854.15  4944.4 1853.02
  4972.7 1847.06  4986.9 1843.17  4989.8 1838.05  4990.2 1837.55  5006.2 1838.05
  5055.5 1843.66  5158.1 1843.89  5323.9 1847.42  5821.3 1849.43  6026.4 1854.32
  6048.4 1856.13  6092.5 1864.50  6130.0 1869.42  6272.9 1882.24  6318.7 1891.44
  6364.5 1896.57  6410.3 1904.57  6445.3 1906.72  6490.1 1912.06  6544.6 1913.35
#Mann=3,-1,0
  3940.4    0.05       0  4989.8    0.05       0  5006.2    0.05       0
Bank Sta=4989.8,5006.2
Exp/Cntr=0.3,0.1

Type RM Length L Ch R = 1,152812,419,419,419
BEGIN DESCRIPTION:
Deadman Creek 191.0
END DESCRIPTION:
XS GIS Cut Line= 3
      1640755.00      6851188.00      1641505.00      6851988.00
      1642905.01      6852188.00
#Sta/Elev= 30
  3902.6 1889.11  4143.2 1871.85  4157.3 1873.53  4171.5 1869.96  4185.6 1868.45
  4348.3 1862.54  4702.0 1852.86  4892.9 1841.85  4942.8 1841.47  4949.6 1839.22
  4987.9 1835.63  4988.3 1835.13  5004.4 1835.63  5009.3 1839.24  5019.4 1838.11
  5029.5 1840.47  5090.1 1840.59  5150.7 1844.67  5645.7 1847.00  5827.5 1851.92
  5857.8 1854.91  5918.4 1865.10  5958.8 1869.36  6019.4 1873.92  6029.5 1876.06
  6140.7 1882.09  6160.9 1884.90  6171.0 1887.90  6201.3 1891.68  6413.4 1911.37
#Mann=3,-1,0
  3902.6    0.05       0  4987.9    0.05       0  5004.4    0.05       0
Bank Sta=4987.9,5004.4
Exp/Cntr=0.3,0.1

Type RM Length L Ch R = 1,152393,242,242,242
BEGIN DESCRIPTION:
Deadman Creek 190.0
END DESCRIPTION:
XS GIS Cut Line= 3
      1640605.03      6851688.02      1641481.97      6852371.53
      1642600.85      6852444.39
#Sta/Elev= 30
  3895.1 1867.69  3916.8 1867.64  4037.1 1860.55  4244.3 1855.67  4457.8 1848.47
  4656.8 1845.27  4785.3 1839.69  4857.6 1841.64  4913.7 1839.84  4978.0 1840.26
  4998.8 1833.80  5016.9 1832.87  5017.4 1832.37  5037.6 1832.87  5040.0 1836.36
  5050.1 1840.26  5080.1 1843.08  5488.6 1844.88  5645.7 1847.70  5691.4 1851.48
  5802.9 1856.89  5821.7 1860.04  5831.7 1864.63  5841.7 1864.04  5851.8 1860.75
  5871.8 1859.69  5950.0 1870.90  5992.1 1874.44  6072.2 1878.10  6128.2 1884.36
#Mann=3,-1,0
  3895.1    0.05       0  5016.9    0.05       0  5037.6    0.05       0
Bank Sta=5016.9,5037.6
Exp/Cntr=0.3,0.1

Type RM Length L Ch R = 1,152151,217,217,217
BEGIN DESCRIPTION:
Mapping XS de6c9c38
END DESCRIPTION:
XS GIS Cut Line= 4
      1640244.64      6851955.58      1640916.48      6852419.10
      1641312.31      6852564.93      1642484.21      6852606.60
#Sta/Elev= 30
  3719.6 1853.22  3729.4 1854.15  3735.5 1852.75  3756.5 1853.61  3786.2 1852.42
  3908.6 1854.11  4347.4 1845.59  4404.1 1845.79  4806.7 1838.89  4867.6 1839.40
  4892.7 1842.58  4898.1 1840.96  4923.2 1838.41  4928.6 1835.39  4948.3 1831.39
  4960.0 1831.34  4960.5 1830.84  4980.7 1831.34  5020.4 1831.81  5050.4 1841.55
  5070.4 1842.52  5140.5 1843.11  5170.5 1841.50  5570.7 1843.81  5720.8 1847.49
  5770.9 1849.65  5850.9 1857.57  5961.0 1862.47  6027.5 1868.74  6130.3 1872.02
#Mann=3,-1,0
  3719.6    0.05       0  4960.0    0.05       0  4980.7    0.05       0
Bank Sta=4960,4980.7
Exp/Cntr=0.3,0.1

Type RM Length L Ch R = 1,151934,286,286,286
BEGIN DESCRIPTION:
Deadman Creek 189.0
END DESCRIPTION:
XS GIS Cut Line= 3
      1640057.09      6852215.97      1641171.69      6852695.14
      1642429.96      6852962.99
#Sta/Elev= 30
  3765.1 1859.15  3804.6 1856.27  3909.6 1852.31  3956.7 1846.88  3991.4 1844.99
  4009.3 1847.76  4032.8 1848.68  4266.5 1845.87  4389.6 1846.28  4503.0 1845.49
  4633.6 1843.02  4793.6 1841.43  4905.7 1837.69  4969.3 1838.43  4974.7 1837.04
  5002.2 1835.30  5006.4 1834.03  5006.9 1833.53  5027.1 1834.03  5032.8 1835.93
  5043.1 1836.70  5110.8 1837.77  5124.9 1838.79  5298.7 1839.51  5497.2 1841.69
  5574.7 1843.54  5901.9 1847.63  6055.2 1851.22  6177.9 1852.26  6264.8 1854.03
#Mann=3,-1,0
  3765.1    0.05       0  5006.4    0.05       0  5027.1    0.05       0
Bank Sta=5006.4,5027.1
Exp/Cntr=0.3,0.1

Type RM Length L Ch R = 1,151648,477,477,477
BEGIN DESCRIPTION:
Mapping XS d775804b
END DESCRIPTION:
XS GIS Cut Line= 4
      1640072.72      6852413.89      1640833.15      6852861.81
      1641406.06      6853064.93      1642170.80      6853200.19
#Sta/Elev= 30
  3846.1 1859.47  3902.2 1855.43  4046.6 1851.08  4083.7 1849.05  4099.4 1847.11
  4142.3 1843.89  4185.3 1842.22  4216.5 1841.99  4259.4 1843.64  4275.1 1843.34
  4333.7 1844.88  4675.2 1842.67  4783.7 1840.09  4836.7 1837.27  4857.9 1834.74
  4868.5 1834.53  4883.1 1834.85  4900.4 1837.13  4944.9 1838.42  4953.4 1835.78
  4970.5 1833.32  5016.5 1831.82  5017.0 1831.32  5037.3 1831.82  5038.3 1833.05
  5048.9 1833.37  5080.7 1837.52  5155.7 1839.38  5500.3 1841.76  6113.1 1850.02
#Mann=3,-1,0
  3846.1    0.05       0  5016.5    0.05       0  5037.3    0.05       0
Bank Sta=5016.5,5037.3
Exp/Cntr=0.3,0.1

Type RM Length L Ch R = 1,151171,588,588,588
BEGIN DESCRIPTION:
Deadman Creek 188.0
END DESCRIPTION:
XS GIS Cut Line= 3
      1640490.00      6852753.98      1640955.00      6853388.00
      1641510.84      6853403.02
#Sta/Elev= 30
  4208.2 1843.21  4257.8 1842.82  4278.6 1843.42  4287.1 1842.92  4429.1 1842.23
  4558.7 1840.49  4679.9 1838.06  4715.4 1836.87  4758.8 1834.40  4836.6 1836.63
  4901.5 1837.03  4916.1 1836.19  4922.3 1834.66  4937.0 1833.57  4951.6 1833.34
  4966.3 1834.12  4980.9 1832.49  4984.8 1829.46  4985.2 1828.96  5001.0 1828.96
  5001.4 1829.46  5034.5 1832.94  5054.5 1836.02  5064.5 1835.67  5074.5 1836.98
  5084.5 1837.32  5114.5 1837.20  5134.5 1836.43  5404.6 1838.89  5550.5 1840.87
#Mann=3,-1,0
  4208.2    0.05       0  4984.8    0.05       0  5001.4    0.05       0
Bank Sta=4984.8,5001.4
Exp/Cntr=0.3,0.1

Type RM Length L Ch R = 1,150583,504,504,504
BEGIN DESCRIPTION:
Mapping XS 5685a17e
END DESCRIPTION:
XS GIS Cut Line= 3
      1640044.48      6853256.96      1640617.39      6853751.74
      1641153.81      6853918.39
#Sta/Elev= 30
  4402.2 1863.53  4410.5 1862.18  4417.1 1862.49  4424.7 1860.73  4431.3 1860.87
  4453.2 1857.44  4459.8 1857.66  4481.7 1854.64  4488.4 1854.74  4502.6 1851.41
  4559.6 1845.87  4580.5 1844.85  4594.8 1842.83  4799.9 1835.78  4864.6 1834.60
  4956.7 1834.98  4971.0 1833.00  4973.7 1828.19  4974.2 1827.69  4994.8 1828.19
  4998.5 1829.83  5027.0 1830.10  5063.1 1832.23  5098.2 1832.34  5141.0 1834.50
  5195.2 1833.96  5298.2 1835.41  5303.4 1834.74  5355.6 1836.15  5720.9 1838.78
#Mann=3,-1,0
  4402.2    0.05       0  4973.7    0.05       0  4994.8    0.05       0
Bank Sta=4973.7,4994.8
Exp/Cntr=0.3,0.1

Type RM Length L Ch R = 1,150079,542,542,542
BEGIN DESCRIPTION:
Deadman Creek 186.0
END DESCRIPTION:
XS GIS Cut Line= 3
      1639804.99      6853788.00      1640155.00      6853988.00
      1641705.02      6855088.01
#Sta/Elev= 30
  4595.7 1887.90  4641.1 1886.82  4749.0 1874.26  4764.9 1870.82  4823.9 1862.84
  4837.6 1858.73  4867.1 1845.41  4904.5 1833.84  4918.2 1831.49  4941.2 1833.32
  4963.5 1832.93  4985.1 1829.16  4995.9 1825.20  5001.9 1825.20  5006.2 1822.99
  5014.0 1821.71  5014.5 1821.21  5040.2 1821.71  5041.9 1825.81  5048.0 1825.38
  5071.4 1831.36  5113.2 1832.93  5543.8 1833.35  5959.6 1838.31  6283.2 1845.32
  6339.7 1847.19  6425.8 1854.39  6633.7 1862.70  6820.7 1873.77  6899.5 1876.92
#Mann=3,-1,0
  4595.7    0.05       0  5014.0    0.05       0  5040.2    0.05       0
Bank Sta=5014,5040.2
Exp/Cntr=0.3,0.1

Type RM Length L Ch R = 1,149537,534,534,534
BEGIN DESCRIPTION:
Deadman Creek 185.0
END DESCRIPTION:
XS GIS Cut Line= 3
      1639700.71      6854277.77      1639905.00      6854438.00
      1641357.00      6855501.76
#Sta/Elev= 30
  4739.4 1865.18  4770.3 1862.20  4828.2 1853.13  4834.5 1851.72  4871.5 1839.14
  4906.8 1830.60  4927.6 1827.60  4962.9 1828.44  4977.3 1827.79  4985.4 1826.35
  4987.9 1823.35  4988.2 1822.85  5005.9 1822.85  5006.2 1823.35  5012.6 1824.97
  5048.6 1827.13  5085.8 1831.30  5127.6 1830.44  5399.3 1831.07  5715.0 1833.58
  5886.4 1836.42  6015.5 1840.48  6107.9 1842.50  6480.0 1849.07  6494.7 1850.09
  6515.5 1849.75  6559.5 1851.19  6666.0 1852.73  6695.4 1854.04  6799.0 1855.90
#Mann=3,-1,0
  4739.4    0.05       0  4987.9    0.05       0  5006.2    0.05       0
Bank Sta=4987.9,5006.2
Exp/Cntr=0.3,0.1

Type RM Length L Ch R = 1,149003,508,508,508
BEGIN DESCRIPTION:
Deadman Creek 184.0
END DESCRIPTION:
XS GIS Cut Line= 3
      1639504.99      6854487.98      1639655.00      6854888.00
      1641054.99      6856287.99
#Sta/Elev= 30
  4566.2 1859.95  4611.6 1856.02  4683.7 1846.60  4727.3 1831.90  4752.2 1828.47
  4769.1 1827.00  4790.5 1826.92  4837.7 1828.94  4886.6 1829.13  4917.8 1826.70
  4940.0 1827.41  4961.4 1826.47  4978.3 1825.07  4983.6 1822.81  4995.5 1821.03
  4995.9 1820.53  5016.6 1821.03  5021.7 1824.60  5035.8 1828.99  5050.0 1829.26
  5290.4 1827.98  5629.8 1831.04  5940.9 1835.83  6138.9 1840.42  6266.2 1846.12
  6534.9 1865.58  6648.0 1870.90  6803.6 1876.47  6888.5 1880.85  6973.3 1881.98
#Mann=3,-1,0
  4566.2    0.05       0  4995.5    0.05       0  5016.6    0.05       0
Bank Sta=4995.5,5016.6
Exp/Cntr=0.3,0.1

Type RM Length L Ch R = 1,148495,573,573,573
BEGIN DESCRIPTION:
Deadman Creek 183.0
END DESCRIPTION:
XS GIS Cut Line= 3
      1638846.30      6854707.54      1639255.00      6855088.00
      1640804.97      6856187.98
#Sta/Elev= 30
  4441.0 1834.43  4758.8 1830.08  4850.6 1826.70  4893.1 1828.42  4914.6 1827.35
  4949.8 1823.17  4985.5 1825.17  5002.4 1824.77  5012.9 1821.83  5042.4 1820.78
  5043.9 1819.59  5044.4 1819.09  5070.5 1819.59  5072.0 1825.89  5078.1 1828.34
  5085.2 1828.44  5229.4 1827.52  5265.1 1824.78  5351.2 1825.99  5379.5 1825.17
  5452.1 1827.10  5924.5 1830.52  6218.5 1835.59  6376.0 1841.47  6533.4 1855.05
  6655.2 1862.71  6678.6 1865.95  6800.4 1867.52  6836.1 1870.26  6900.0 1871.65
#Mann=3,-1,0
  4441.0    0.05       0  5043.9    0.05       0  5070.5    0.05       0
Bank Sta=5043.9,5070.5
Exp/Cntr=0.3,0.1

Type RM Length L Ch R = 1,147922,933,933,933
BEGIN DESCRIPTION:
Deadman Creek 182.0
END DESCRIPTION:
XS GIS Cut Line= 3
      1638505.02      6855388.00      1639005.00      6855388.00
      1640555.04      6856188.02
#Sta/Elev= 30
  4500.8 1847.30  4690.8 1836.70  4750.8 1827.54  4820.8 1826.39  4860.8 1824.56
  4890.8 1825.67  4930.8 1822.26  4980.8 1821.72  4990.8 1818.79  4991.0 1817.72
  4991.5 1817.22  5014.9 1817.72  5031.2 1823.99  5036.8 1822.21  5045.8 1825.53
  5075.5 1825.39  5097.7 1826.64  5252.7 1825.10  5297.1 1825.93  5327.1 1824.73
  5341.4 1825.26  5380.1 1823.33  5529.5 1826.42  6011.3 1830.16  6299.3 1835.34
  6365.8 1838.00  6486.2 1847.61  6543.0 1853.27  6610.0 1857.73  6745.1 1863.87
#Mann=3,-1,0
  4500.8    0.05       0  4991.0    0.05       0  5014.9    0.05       0
Bank Sta=4991,5014.9
Exp/Cntr=0.3,0.1

Type RM Length L Ch R = 1,146989,690,690,690
BEGIN DESCRIPTION:
Deadman Creek 181.0
END DESCRIPTION:
XS GIS Cut Line= 3
      1638289.43      6855632.67      1639218.56      6856106.60
      1640071.39      6856595.41
#Sta/Elev= 30
  3903.8 1854.18  3921.1 1853.75  4022.3 1845.91  4044.8 1845.12  4157.0 1834.01
  4269.3 1824.88  4304.6 1823.96  4560.1 1824.40  4707.1 1822.33  4752.0 1823.46
  4841.8 1822.21  4871.4 1823.16  4915.8 1821.24  4946.8 1821.23  4965.8 1819.78
  4981.4 1820.14  4997.2 1819.05  5018.8 1816.22  5021.2 1814.89  5021.7 1814.39
  5048.0 1814.89  5062.0 1821.08  5077.8 1823.88  5282.1 1826.23  5604.3 1832.84
  5765.5 1836.97  5772.6 1838.16  5808.6 1838.43  5905.0 1842.32  5929.8 1844.10
#Mann=3,-1,0
  3903.8    0.05       0  5021.2    0.05       0  5048.0    0.05       0
Bank Sta=5021.2,5048
Exp/Cntr=0.3,0.1

Type RM Length L Ch R = 1,146299,567,567,567
BEGIN DESCRIPTION:
Deadman Creek 180.0
END DESCRIPTION:
XS GIS Cut Line= 3
      1638005.03      6855788.02      1638755.00      6856238.00
      1640755.01      6857438.00
#Sta/Elev= 30
  4130.8 1868.67  4189.1 1862.40  4422.3 1844.43  4589.5 1824.04  4678.9 1822.64
  4912.1 1823.56  4939.3 1820.33  4947.1 1817.44  4991.3 1812.08  4991.7 1811.58
  5012.7 1812.08  5040.4 1820.03  5055.9 1820.81  5087.0 1819.91  5129.8 1821.73
  5304.7 1822.76  5646.8 1822.29  5872.3 1826.05  6126.9 1832.83  6222.1 1837.95
  6360.1 1850.97  6521.5 1862.83  6593.4 1865.14  6603.1 1867.64  6638.1 1869.34
  6645.9 1871.13  6651.7 1870.05  6848.0 1872.81  7149.3 1879.54  7337.8 1876.05
#Mann=3,-1,0
  4130.8    0.05       0  4991.3    0.05       0  5012.7    0.05       0
Bank Sta=4991.3,5012.7
Exp/Cntr=0.3,0.1

Type RM Length L Ch R = 1,145732,485,485,485
BEGIN DESCRIPTION:
Deadman Creek 179.0
END DESCRIPTION:
XS GIS Cut Line= 3
      1637754.99      6856338.00      1638455.00      6856688.00
      1640005.04      6857038.01
#Sta/Elev= 30
  4213.3 1866.12  4302.8 1858.18  4473.3 1840.56  4504.0 1836.59  4557.1 1822.69
  4579.5 1820.95  4674.5 1820.06  4959.6 1821.04  4982.0 1813.13  4987.5 1813.91
  4993.1 1811.79  4993.4 1810.68  4993.9 1810.18  5017.6 1810.68  5020.1 1810.76
  5026.7 1814.52  5057.4 1815.44  5077.9 1818.92  5106.5 1820.49  5170.2 1818.98
  5252.2 1820.87  5521.0 1819.28  5764.8 1820.65  5973.5 1824.05  6205.6 1830.64
  6256.9 1833.54  6369.7 1842.87  6390.2 1845.66  6469.3 1852.46  6585.0 1859.62
#Mann=3,-1,0
  4213.3    0.05       0  4993.4    0.05       0  5017.6    0.05       0
Bank Sta=4993.4,5017.6
Exp/Cntr=0.3,0.1

Type RM Length L Ch R = 1,145247,860,860,860
BEGIN DESCRIPTION:
Deadman Creek 178.0
END DESCRIPTION:
XS GIS Cut Line= 3
      1637624.69      6857119.16      1638424.13      6857159.58
      1640005.03      6857138.00
#Sta/Elev= 30
  4219.1 1852.68  4269.5 1848.72  4389.6 1836.12  4469.7 1830.12  4509.8 1822.76
  4539.8 1819.96  4609.9 1818.41  4688.1 1814.21  4750.1 1816.94  4960.4 1819.18
  4990.4 1815.58  4997.3 1809.22  4997.8 1808.72  5021.5 1809.22  5022.5 1810.73
  5030.4 1812.85  5050.4 1813.15  5080.4 1817.60  5120.4 1818.97  5350.5 1817.75
  5450.5 1815.51  5530.5 1818.13  5810.5 1820.49  6110.5 1826.36  6160.5 1829.11
  6200.5 1833.84  6234.9 1835.88  6310.5 1845.16  6380.6 1851.91  6600.6 1862.88
#Mann=3,-1,0
  4219.1    0.05       0  4997.3    0.05       0  5021.5    0.05       0
Bank Sta=4997.3,5021.5
Exp/Cntr=0.3,0.1

Type RM Length L Ch R = 1,144387,346,346,346
BEGIN DESCRIPTION:
Mapping XS 59463c89
END DESCRIPTION:
XS GIS Cut Line= 3
      1637422.65      6857604.19      1638437.60      6857608.68
      1639650.33      6857604.33
#Sta/Elev= 30
  3716.8 1853.69  3749.2 1850.79  3799.2 1848.10  3829.2 1841.22  3859.2 1840.48
  3869.2 1839.52  3899.2 1833.69  3939.2 1831.25  3959.2 1829.00  3979.2 1823.12
  3999.2 1819.21  4059.2 1816.39  4259.2 1813.40  4309.2 1810.70  4369.2 1814.20
  4539.2 1816.95  4929.2 1816.31  4939.2 1815.23  4969.2 1809.35  4985.7 1808.91
  4986.2 1808.41  5012.7 1808.91  5019.2 1810.81  5039.2 1812.54  5119.2 1812.73
  5189.2 1816.23  5619.2 1821.31  5739.2 1824.21  5829.2 1827.77  5944.5 1836.50
#Mann=3,-1,0
  3716.8    0.05       0  4985.7    0.05       0  5012.7    0.05       0
Bank Sta=4985.7,5012.7
Exp/Cntr=0.3,0.1

Type RM Length L Ch R = 1,144041,678,678,678
BEGIN DESCRIPTION:
Deadman Creek 177.0
END DESCRIPTION:
XS GIS Cut Line= 4
      1637436.08      6857729.94      1638328.76      6857724.69
      1638655.00      6857938.00      1639455.03      6858688.02
#Sta/Elev= 30
  3722.4 1848.71  3761.3 1844.48  3811.3 1836.46  3841.3 1834.09  3881.3 1828.92
  3921.3 1820.31  3941.3 1817.97  3971.3 1816.56  4231.3 1812.42  4271.3 1810.39
  4331.3 1813.39  4451.3 1815.38  4671.6 1815.52  4722.9 1813.17  4774.2 1814.54
  4837.6 1814.25  4940.0 1811.41  4989.8 1807.75  4990.2 1807.25  5013.3 1807.75
  5026.1 1811.08  5047.1 1814.37  5068.6 1815.65  5549.7 1821.14  5684.1 1818.97
  5775.9 1820.10  5931.7 1826.37  5974.2 1827.02  6045.0 1831.94  6101.5 1832.89
#Mann=3,-1,0
  3722.4    0.05       0  4989.8    0.05       0  5013.3    0.05       0
Bank Sta=4989.8,5013.3
Exp/Cntr=0.3,0.1

Type RM Length L Ch R = 1,143363,613,613,613
BEGIN DESCRIPTION:
Deadman Creek 176.0
END DESCRIPTION:
XS GIS Cut Line= 4
      1637350.81      6857788.32      1637805.43      6857830.12
      1638430.16      6858285.87      1639455.00      6859538.00
#Sta/Elev= 30
  4180.1 1854.37  4235.4 1850.48  4274.7 1845.26  4375.1 1830.74  4395.2 1825.14
  4415.3 1823.27  4435.4 1817.46  4455.4 1815.72  4648.5 1813.53  4727.7 1808.01
  4878.3 1812.70  4957.8 1813.12  4970.3 1810.94  4983.0 1803.78  4983.4 1803.28
  5006.5 1803.78  5020.4 1808.96  5093.8 1810.19  5143.6 1813.32  5185.7 1811.28
  5265.3 1813.25  5451.0 1813.68  5606.5 1817.59  6417.2 1828.62  6481.1 1831.19
  6537.0 1836.62  6629.6 1842.51  6878.7 1850.71  6907.4 1853.06  7028.0 1855.35
#Mann=3,-1,0
  4180.1    0.05       0  4983.0    0.03       0  5006.5    0.05       0
Bank Sta=4983,5006.5
Exp/Cntr=0.3,0.1

Type RM Length L Ch R = 1,142750,614,614,614
BEGIN DESCRIPTION:
Deadman Creek 175.0
END DESCRIPTION:
XS GIS Cut Line= 3
      1637334.35      6857898.32      1638243.07      6858553.14
      1639054.97      6859187.98
#Sta/Elev= 30
  3864.9 1854.33  3908.0 1851.81  3922.7 1849.07  3979.2 1842.62  4029.5 1831.64
  4044.2 1826.35  4073.6 1819.49  4094.5 1817.06  4159.5 1812.99  4245.4 1811.36
  4281.0 1809.81  4287.2 1808.54  4322.8 1807.68  4366.9 1810.77  4423.4 1811.86
  4666.9 1812.94  4897.1 1811.50  4925.7 1810.43  4962.1 1806.84  4980.5 1802.66
  4980.9 1802.16  5006.9 1802.66  5011.8 1806.14  5018.2 1807.16  5025.5 1810.70
  5032.6 1812.61  5076.0 1814.41  5780.5 1824.45  5965.0 1828.72  6015.6 1832.21
#Mann=3,-1,0
  3864.9    0.05       0  4980.5    0.05       0  5006.9    0.05       0
Bank Sta=4980.5,5006.9
Exp/Cntr=0.3,0.1

Type RM Length L Ch R = 1,142136,322,322,322
BEGIN DESCRIPTION:
Deadman Creek 174.0
END DESCRIPTION:
XS GIS Cut Line= 3
      1637227.43      6858103.21      1637810.99      6858615.50
      1639255.00      6860088.00
#Sta/Elev= 30
  4262.8 1858.37  4384.9 1853.60  4434.2 1847.29  4462.7 1841.53  4470.3 1837.41
  4505.4 1827.60  4519.6 1821.58  4576.5 1813.06  4597.4 1811.46  4654.3 1811.41
  4668.6 1807.65  4689.5 1806.17  4760.6 1809.70  4959.0 1810.31  4972.7 1800.99
  4973.2 1800.49  5002.1 1800.99  5008.3 1804.35  5015.9 1803.81  5022.5 1806.62
  5065.2 1807.68  5270.2 1806.68  5355.0 1811.42  5439.9 1813.21  5963.2 1818.09
  6422.9 1830.70  6620.9 1843.57  6741.0 1855.54  7045.2 1878.96  7101.7 1881.25
#Mann=3,-1,0
  4262.8    0.05       0  4972.7    0.05       0  5002.1    0.05       0
Bank Sta=4972.7,5002.1
Exp/Cntr=0.3,0.1

Type RM Length L Ch R = 1,141814,499,499,499
BEGIN DESCRIPTION:
Deadman Creek 173.0
END DESCRIPTION:
XS GIS Cut Line= 3
      1637205.02      6858438.02      1637530.42      6858771.84
      1639104.99      6860137.99
#Sta/Elev= 30
  4540.5 1854.25  4618.3 1845.85  4660.7 1835.04  4681.8 1825.76  4710.1 1816.83
  4780.9 1806.23  4809.2 1804.35  4865.7 1808.27  4986.1 1810.18  5000.2 1805.72
  5006.4 1801.93  5006.8 1799.75  5007.3 1799.25  5036.3 1799.75  5050.0 1806.03
  5085.2 1807.29  5127.9 1807.76  5148.8 1805.54  5277.0 1808.66  5304.5 1805.98
  5333.0 1811.19  5354.9 1812.02  5864.8 1814.49  6028.2 1816.94  6509.6 1830.06
  6552.4 1831.76  6722.3 1844.52  6807.8 1853.52  7027.2 1870.75  7091.3 1877.91
#Mann=3,-1,0
  4540.5    0.05       0  5006.8    0.05       0  5036.3    0.05       0
Bank Sta=5006.8,5036.3
Exp/Cntr=0.3,0.1

Type RM Length L Ch R = 1,141315,913,913,913
BEGIN DESCRIPTION:
Deadman Creek 172.0
END DESCRIPTION:
XS GIS Cut Line= 3
      1637105.01      6858738.01      1637405.00      6859188.00
      1638805.04      6860438.03
#Sta/Elev= 30
  4464.8 1836.03  4487.3 1830.18  4523.4 1818.08  4580.5 1810.82  4595.5 1807.71
  4609.0 1802.77  4622.5 1800.45  4645.1 1800.36  4694.6 1807.61  4832.9 1808.59
  4905.0 1806.97  4926.0 1803.07  4947.0 1801.53  4947.3 1799.10  4947.8 1798.60
  4976.8 1799.10  4992.1 1799.57  5009.0 1802.12  5019.4 1807.02  5041.1 1808.12
  5770.2 1813.36  5990.0 1817.19  6259.2 1824.96  6308.5 1827.75  6358.7 1833.58
  6493.3 1843.89  6577.7 1853.31  6769.2 1868.16  6832.7 1875.81  6882.5 1878.80
#Mann=3,-1,0
  4464.8    0.05       0  4947.3    0.05       0  4976.8    0.05       0
Bank Sta=4947.3,4976.8
Exp/Cntr=0.3,0.1

Type RM Length L Ch R = 1,140402,200,200,200
BEGIN DESCRIPTION:
Mapping XS 062d10f5
END DESCRIPTION:
XS GIS Cut Line= 6
      1637010.23      6858773.26      1636916.48      6859049.31
      1636890.44      6859367.02      1637025.86      6860424.31
      1637031.06      6860580.56      1637671.67      6861075.33
#Sta/Elev= 30
  3999.2 1835.84  4025.3 1833.73  4030.8 1832.22  4062.2 1828.90  4109.8 1819.98
  4213.9 1809.74  4276.6 1807.89  4281.9 1808.53  4419.9 1802.48  4500.1 1803.01
  4530.2 1805.46  4570.4 1806.03  4892.8 1804.29  4924.5 1802.31  4963.4 1801.87
  4989.4 1797.39  4989.9 1796.89  5019.0 1797.39  5044.0 1803.62  5054.1 1805.40
  5064.2 1805.70  5215.4 1804.92  5789.2 1808.85  6161.0 1815.16  6210.8 1817.66
  6316.9 1828.43  6403.7 1832.41  6524.1 1840.63  6594.9 1844.24  6641.2 1845.09
#Mann=3,-1,0
  3999.2    0.05       0  4989.4    0.05       0  5019.0    0.05       0
Bank Sta=4989.4,5019
Exp/Cntr=0.3,0.1

Type RM Length L Ch R = 1,140202,1059,1059,1059
BEGIN DESCRIPTION:
Mapping XS c33c0f91
END DESCRIPTION:
XS GIS Cut Line= 4
      1636817.53      6858627.40      1636718.56      6859346.18
      1636827.94      6860486.81      1637598.78      6861111.81
#Sta/Elev= 30
  3780.0 1837.31  3942.1 1829.55  3952.2 1828.42  3972.4 1824.16  3984.7 1823.76
  3992.6 1821.98  4022.9 1818.34  4123.6 1810.17  4214.7 1808.01  4587.8 1804.07
  4768.6 1804.13  4848.9 1803.02  4889.1 1801.04  4929.3 1801.75  4949.4 1799.60
  4986.3 1798.26  4986.8 1797.76  5013.0 1798.26  5019.7 1801.70  5044.6 1805.45
  5220.6 1803.27  5291.0 1804.50  5678.5 1806.37  6162.6 1814.43  6212.3 1816.78
  6282.7 1825.42  6332.3 1828.76  6418.5 1833.07  6574.6 1843.92  6643.8 1845.88
#Mann=3,-1,0
  3780.0    0.05       0  4986.3    0.05       0  5013.0    0.05       0
Bank Sta=4986.3,5013
Exp/Cntr=0.3,0.1

Type RM Length L Ch R = 1,139143,1019,1019,1019
BEGIN DESCRIPTION:
Deadman Creek 170.0
END DESCRIPTION:
XS GIS Cut Line= 3
      1635705.05      6859838.01      1636105.00      6859938.00
      1637655.00      6861188.00
#Sta/Elev= 30
  4575.3 1852.51  4639.7 1848.81  4680.9 1834.15  4729.9 1812.57  4758.2 1805.27
  4781.4 1803.41  4936.0 1802.14  4956.6 1797.98  4977.3 1796.62  4994.8 1793.70
  5093.9 1797.29  5116.0 1795.66  5126.4 1793.43  5127.1 1792.93  5160.7 1793.43
  5165.9 1798.17  5172.3 1797.50  5193.1 1800.36  5229.9 1801.77  5393.0 1802.86
  5527.4 1800.18  5628.1 1803.80  6018.4 1807.40  6410.2 1814.58  6459.8 1818.38
  6488.6 1822.51  6544.6 1827.31  6666.1 1833.94  6800.5 1843.42  6978.8 1849.76
#Mann=3,-1,0
  4575.3    0.05       0  5126.4    0.05       0  5160.7    0.05       0
Bank Sta=5126.4,5160.7
Exp/Cntr=0.3,0.1

Type RM Length L Ch R = 1,138124,472,472,472
BEGIN DESCRIPTION:
Deadman Creek 169.0
END DESCRIPTION:
XS GIS Cut Line= 3
      1635655.01      6859988.02      1636361.07      6860779.85
      1637105.02      6861438.01
#Sta/Elev= 30
  3939.1 1850.02  4009.7 1843.57  4023.9 1838.55  4038.2 1831.66  4101.7 1809.65
  4166.1 1799.88  4215.4 1798.69  4342.5 1801.33  4477.1 1801.60  4888.4 1799.29
  4909.3 1797.06  4958.7 1797.06  4972.9 1793.70  4980.4 1789.13  4981.9 1786.58
  4982.5 1786.08  5009.4 1786.58  5022.6 1791.44  5030.1 1792.50  5051.0 1800.20
  5065.2 1803.31  5079.5 1802.62  5086.1 1804.62  5575.5 1813.48  5653.3 1819.94
  5823.1 1827.88  5830.6 1829.48  5873.1 1831.35  5879.9 1832.74  5993.3 1838.81
#Mann=3,-1,0
  3939.1    0.05       0  4981.9    0.05       0  5009.4    0.05       0
#XS Ineff=2,0
    0.00 4700.00 1809.04               0
Permanent Ineff=
       F       F
Bank Sta=4981.9,5009.4
Exp/Cntr=0.3,0.1

Type RM Length L Ch R = 1,137652,610,610,610
BEGIN DESCRIPTION:
Deadman Creek 168.0
END DESCRIPTION:
XS GIS Cut Line= 3
      1635555.02      6860088.04      1635947.72      6860937.79
      1636555.00      6861688.00
#Sta/Elev= 30
  4063.9 1845.36  4101.0 1840.44  4141.0 1831.18  4146.9 1828.34  4163.0 1823.77
  4169.8 1820.90  4207.1 1810.26  4273.2 1797.94  4290.0 1797.09  4318.4 1799.55
  4350.3 1799.98  4779.9 1799.55  4846.0 1795.81  4923.1 1794.98  4931.3 1792.51
  4974.8 1786.40  4975.4 1785.90  5005.9 1786.40  5013.1 1793.35  5019.5 1794.59
  5026.0 1797.96  5040.4 1797.79  5141.0 1801.71  5360.5 1805.17  5411.2 1806.87
  5502.4 1807.69  5708.6 1812.65  5780.5 1815.36  5850.9 1820.83  5965.2 1827.40
#Mann=3,-1,0
  4063.9    0.05       0  4974.8    0.05       0  5005.9    0.05       0
#XS Ineff=2,0
    0.00 4706.40 1810.74               0
Permanent Ineff=
       F       F
Bank Sta=4974.8,5005.9
Exp/Cntr=0.3,0.1

Type RM Length L Ch R = 1,137042,653,653,653
BEGIN DESCRIPTION:
Deadman Creek 167.0
END DESCRIPTION:
XS GIS Cut Line= 3
      1635055.00      6860388.01      1635466.30      6861113.96
      1635987.11      6861843.09
#Sta/Elev= 30
  4155.3 1818.18  4190.6 1813.50  4235.7 1803.19  4265.7 1800.77  4384.0 1798.60
  4557.6 1797.40  4588.9 1795.02  4661.0 1798.15  4948.3 1799.14  4971.2 1797.94
  4977.0 1791.08  4982.8 1788.11  4996.3 1785.30  4996.9 1784.80  5027.4 1785.30
  5056.1 1792.49  5069.7 1793.43  5142.1 1794.35  5199.9 1793.09  5228.1 1794.52
  5256.5 1797.49  5523.1 1805.23  5615.3 1809.19  5701.3 1810.18  5781.1 1813.12
  5787.4 1814.38  5823.0 1814.34  5837.7 1815.55  5843.9 1814.74  5885.7 1817.42
#Mann=3,-1,0
  4155.3    0.05       0  4996.3    0.03       0  5027.4    0.05       0
#XS Ineff=2,0
    0.00 4883.30 1805.24               0
Permanent Ineff=
       F       F
Bank Sta=4996.3,5027.4
Exp/Cntr=0.3,0.1

Type RM Length L Ch R = 1,136389,625,625,625
BEGIN DESCRIPTION:
Deadman Creek 166.0
END DESCRIPTION:
XS GIS Cut Line= 3
      1633950.65      6860561.85      1635105.00      6861638.00
      1635398.60      6861999.39
#Sta/Elev= 30
  3427.2 1829.83  3484.3 1827.82  3541.0 1824.04  3604.5 1816.50  3653.8 1809.20
  3675.3 1808.17  3724.6 1802.58  3880.5 1798.24  3923.0 1796.50  3965.5 1792.87
  4029.0 1794.62  4149.2 1795.45  4835.6 1796.53  4870.8 1795.63  4892.3 1792.03
  4906.4 1787.10  4913.3 1786.37  4941.6 1788.87  4955.8 1786.90  4984.1 1789.21
  4991.5 1786.40  4992.4 1783.60  4992.7 1783.10  5009.6 1783.60  5019.0 1787.88
  5033.4 1788.40  5055.7 1792.27  5134.0 1794.12  5317.8 1802.93  5471.0 1816.52
#Mann=3,-1,0
  3427.2    0.05       0  4992.4    0.05       0  5009.6    0.05       0
#XS Ineff=2,0
    0.00 4716.90 1805.42               0
Permanent Ineff=
       F       F
Bank Sta=4992.4,5009.6
Exp/Cntr=0.3,0.1

Type RM Length L Ch R = 1,135764,812,812,812
BEGIN DESCRIPTION:
Deadman Creek 165.0
END DESCRIPTION:
XS GIS Cut Line= 3
      1634009.50      6861336.18      1634728.06      6862086.18
      1635005.01      6862388.01
#Sta/Elev= 30
  3959.4 1796.41  4403.2 1793.06  4474.0 1789.65  4502.0 1790.86  4537.5 1793.84
  4551.6 1793.53  4601.0 1795.05  4685.9 1793.11  4735.6 1790.94  4905.1 1791.41
  4919.3 1790.53  4940.7 1787.28  4969.0 1785.79  4975.9 1784.14  4989.4 1778.55
  4990.1 1778.05  5017.1 1778.55  5018.3 1781.10  5025.7 1786.79  5032.5 1788.67
  5039.9 1792.82  5046.7 1792.61  5060.9 1793.95  5145.9 1793.99  5188.5 1796.02
  5216.9 1801.29  5237.8 1807.69  5252.0 1810.06  5365.5 1822.65  5407.7 1825.98
#Mann=3,-1,0
  3959.4    0.05       0  4989.4    0.05       0  5017.1    0.05       0
#XS Ineff=2,0
    0.00 4583.70 1803.45               0
Permanent Ineff=
       F       F
Bank Sta=4989.4,5017.1
Exp/Cntr=0.3,0.1

Type RM Length L Ch R = 1,134952,540,540,540
BEGIN DESCRIPTION:
Deadman Creek 164.0
END DESCRIPTION:
XS GIS Cut Line= 3
      1633412.23      6861560.76      1634045.43      6862297.25
      1634755.03      6862538.01
#Sta/Elev= 30
  4099.6 1802.92  4504.3 1794.71  4709.5 1787.44  4787.4 1791.54  4844.4 1792.38
  4908.1 1791.41  4922.3 1789.44  4928.9 1786.82  4936.6 1786.36  4943.2 1783.39
  4950.9 1782.31  4954.4 1779.97  4955.2 1779.47  4989.0 1779.97  4992.7 1782.86
  5000.3 1781.93  5014.5 1782.56  5092.8 1787.39  5133.8 1788.11  5165.5 1787.19
  5181.7 1788.31  5250.1 1789.09  5342.5 1791.02  5640.6 1792.23  5693.4 1793.48
  5704.0 1794.38  5735.7 1801.50  5741.7 1805.41  5746.9 1806.65  5820.2 1816.18
#Mann=5,-1,0
  4099.6    0.05       0  4954.4    0.03       0  4989.0    0.05       0
  5250.1    0.12       0  5342.5    0.05       0
#XS Ineff=2,0
    0.00 4827.30 1797.00               0
Permanent Ineff=
       F       F
Bank Sta=4954.4,4989
Exp/Cntr=0.3,0.1

Type RM Length L Ch R = 1,134412,141,141,141
BEGIN DESCRIPTION:
Deadman Creek 163.0
END DESCRIPTION:
XS GIS Cut Line= 3
      1632796.96      6862652.04      1634207.11      6862759.82
      1634855.02      6862537.99
#Sta/Elev= 30
  3780.7 1823.50  3999.4 1804.23  4019.4 1800.49  4060.2 1797.63  4321.8 1789.21
  4380.5 1783.76  4447.5 1785.24  4470.7 1783.82  4631.2 1786.01  4671.3 1788.07
  4781.7 1790.00  4892.0 1787.24  4912.0 1785.65  4932.1 1781.40  4964.9 1780.55
  4965.6 1780.05  4999.5 1780.55  5022.4 1781.21  5082.5 1786.38  5106.5 1786.76
  5132.7 1790.17  5274.9 1789.13  5587.8 1793.06  5613.8 1796.91  5619.1 1796.34
  5645.1 1803.65  5650.4 1802.99  5668.4 1807.24  5832.8 1821.27  5879.8 1823.34
#Mann=3,-1,0
  3780.7    0.05       0  4964.9    0.03       0  4999.5    0.05       0
#XS Ineff=2,0
    0.00 4765.10 1797.39               0
Permanent Ineff=
       F       F
Bank Sta=4964.9,4999.5
Exp/Cntr=0.3,0.1

Type RM Length L Ch R = 1,134271,621,621,621
BEGIN DESCRIPTION:
Mapping XS c67fe878
END DESCRIPTION:
XS GIS Cut Line= 3
      1633080.90      6862791.04      1634398.59      6862900.41
      1634810.01      6862660.85
#Sta/Elev= 30
  4022.1 1795.05  4226.9 1789.57  4427.6 1788.57  4538.0 1785.46  4588.1 1782.95
  4618.2 1783.88  4678.4 1788.83  4767.4 1789.04  4818.9 1786.48  4859.1 1786.06
  4879.1 1783.93  4888.1 1781.83  4893.1 1782.41  4939.3 1779.67  4949.4 1781.06
  4989.5 1782.52  4999.6 1782.05  5012.4 1777.98  5013.1 1777.48  5047.0 1777.98
  5049.7 1788.51  5417.0 1791.73  5467.5 1791.14  5571.6 1792.69  5593.2 1794.46
  5620.5 1799.19  5652.0 1802.35  5657.8 1803.80  5753.7 1808.22  5820.4 1814.49
#Mann=3,-1,0
  4022.1    0.05       0  5012.4    0.05       0  5047.0    0.05       0
#XS Ineff=2,0
    0.00 4699.50 1794.18               0
Permanent Ineff=
       F       F
Bank Sta=5012.4,5047
Exp/Cntr=0.3,0.1

Type RM Length L Ch R = 1,133650,705,705,705
BEGIN DESCRIPTION:
Deadman Creek 162.0
END DESCRIPTION:
XS GIS Cut Line= 3
      1632955.01      6862738.01      1633755.00      6863388.00
      1635304.98      6864487.99
#Sta/Elev= 30
  3977.2 1808.54  4033.9 1804.56  4062.7 1799.62  4112.2 1796.44  4126.6 1794.39
  4219.3 1790.18  4332.8 1787.94  4524.5 1787.34  4666.8 1784.15  4716.3 1781.27
  4773.8 1786.63  4815.4 1785.52  4858.6 1781.75  4936.8 1780.40  4954.2 1775.14
  4955.0 1774.64  4989.8 1775.14  5000.8 1782.25  5004.7 1783.42  5044.8 1787.41
  5603.4 1788.35  5695.6 1789.59  5739.9 1791.78  5832.2 1799.49  6019.2 1806.19
  6334.1 1819.99  6449.8 1824.14  6758.5 1831.09  6871.8 1834.41  6908.6 1836.76
#Mann=3,-1,0
  3977.2    0.05       0  4954.2    0.05       0  4989.8    0.05       0
Bank Sta=4954.2,4989.8
Exp/Cntr=0.3,0.1

Type RM Length L Ch R = 1,132945,417,417,417
BEGIN DESCRIPTION:
Deadman Creek 161.0
END DESCRIPTION:
XS GIS Cut Line= 3
      1632605.03      6862838.04      1633169.69      6863572.69
      1633439.16      6864542.77
#Sta/Elev= 30
  4073.5 1835.38  4136.9 1830.49  4244.7 1826.18  4300.9 1821.19  4387.9 1817.55
  4523.0 1808.43  4558.3 1803.94  4622.6 1799.59  4672.5 1791.67  4687.0 1790.80
  4707.8 1785.92  4729.3 1784.10  4936.2 1783.71  4943.7 1783.11  4957.0 1775.36
  4974.4 1774.02  4974.9 1773.52  4997.2 1774.02  5000.1 1776.40  5016.0 1778.06
  5026.4 1778.49  5035.1 1775.82  5047.1 1775.48  5113.9 1779.81  5171.7 1779.51
  5182.0 1778.89  5187.6 1776.81  5244.3 1784.06  5431.1 1786.08  6006.9 1787.14
#Mann=3,-1,0
  4073.5    0.05       0  4974.4    0.05       0  4997.2    0.05       0
Bank Sta=4974.4,4997.2
Exp/Cntr=0.3,0.1

Type RM Length L Ch R = 1,132528,563,563,563
BEGIN DESCRIPTION:
Deadman Creek 160.0
END DESCRIPTION:
XS GIS Cut Line= 3
      1632755.00      6863437.99      1632855.00      6863838.00
      1633336.08      6865192.06
#Sta/Elev= 30
  4592.6 1810.27  4623.5 1808.12  4726.6 1804.50  4780.7 1798.38  4809.1 1796.48
  4858.0 1787.91  4863.2 1785.54  4899.3 1776.82  4922.5 1777.46  4940.5 1775.57
  4974.0 1775.34  4981.7 1773.84  4986.0 1770.69  4986.5 1770.19  5008.7 1770.69
  5015.0 1775.51  5020.3 1775.85  5026.1 1778.62  5045.9 1780.45  5100.4 1779.91
  5280.8 1783.76  5467.2 1783.06  5888.6 1785.85  6055.5 1788.10  6093.9 1789.80
  6150.3 1789.91  6186.5 1791.90  6257.2 1792.47  6342.1 1795.29  6441.9 1796.64
#Mann=3,-1,0
  4592.6    0.05       0  4986.0    0.05       0  5008.7    0.05       0
Bank Sta=4986,5008.7
Exp/Cntr=0.3,0.1

Type RM Length L Ch R = 1,131965,546,546,546
BEGIN DESCRIPTION:
Deadman Creek 159.0
END DESCRIPTION:
XS GIS Cut Line= 3
      1632355.00      6863637.98      1632355.00      6864038.00
      1632830.45      6865367.95
#Sta/Elev= 30
  4600.4 1807.07  4670.4 1803.58  4720.4 1798.24  4770.4 1791.52  4850.4 1786.59
  4930.4 1775.83  4950.4 1773.77  4970.4 1773.68  4980.4 1770.18  4990.1 1769.25
  4990.5 1768.75  5008.3 1769.25  5010.5 1771.29  5021.7 1775.69  5041.3 1775.18
  5064.1 1779.65  5077.4 1780.37  5102.8 1779.56  5195.2 1781.98  5251.5 1782.40
  5517.9 1779.98  5635.7 1780.07  5907.4 1784.25  6086.8 1788.20  6136.7 1790.56
  6168.6 1790.43  6266.2 1793.60  6338.5 1800.46  6384.0 1801.68  6412.8 1803.93
#Mann=3,-1,0
  4600.4    0.05       0  4990.1    0.05       0  5008.3    0.05       0
Bank Sta=4990.1,5008.3
Exp/Cntr=0.3,0.1

Type RM Length L Ch R = 1,131419,572,572,572
BEGIN DESCRIPTION:
Deadman Creek 158.0
END DESCRIPTION:
XS GIS Cut Line= 3
      1632005.00      6863638.01      1631905.00      6864288.00
      1632555.01      6865688.03
#Sta/Elev= 30
  4347.5 1805.38  4438.5 1799.62  4489.1 1793.17  4644.7 1789.59  4671.3 1787.24
  4707.9 1781.22  4752.2 1781.09  4771.2 1777.95  4776.2 1779.16  4792.7 1775.01
  4812.9 1774.10  4844.5 1776.12  4873.6 1773.58  4907.8 1773.22  4944.4 1769.14
  4954.5 1770.38  4976.0 1769.70  4977.3 1766.42  4977.9 1765.92  5004.6 1766.42
  5005.1 1770.45  5042.2 1778.06  5059.6 1778.89  5291.8 1780.13  5556.4 1778.66
  6008.4 1790.63  6105.8 1799.19  6397.1 1813.55  6511.6 1821.36  6548.7 1822.50
#Mann=3,-1,0
  4347.5    0.05       0  4977.3    0.05       0  5004.6    0.05       0
Bank Sta=4977.3,5004.6
Exp/Cntr=0.3,0.1

Type RM Length L Ch R = 1,130847,582,582,582
BEGIN DESCRIPTION:
Deadman Creek 157.0
END DESCRIPTION:
XS GIS Cut Line= 3
      1631422.71      6863262.80      1631455.00      6864588.00
      1631409.23      6865521.78
#Sta/Elev= 30
  3668.2 1807.12  3753.4 1803.47  3793.4 1799.41  3913.5 1790.72  4023.5 1785.86
  4133.5 1783.29  4183.6 1780.80  4273.6 1780.95  4463.6 1778.58  4813.7 1778.50
  4893.8 1777.09  4953.8 1777.99  4996.3 1772.35  5001.1 1765.67  5002.1 1765.17
  5046.6 1765.67  5063.9 1767.01  5073.9 1769.48  5113.9 1768.15  5154.0 1777.71
  5194.0 1776.85  5224.1 1778.25  5284.1 1777.91  5364.2 1773.66  5502.0 1781.12
  5507.0 1780.40  5594.5 1783.43  5754.7 1786.42  5884.9 1793.21  5928.7 1794.09
#Mann=3,-1,0
  3668.2    0.05       0  5001.1    0.05       0  5046.6    0.05       0
Bank Sta=5001.1,5046.6
Exp/Cntr=0.3,0.1

Type RM Length L Ch R = 1,130265,552,552,552
BEGIN DESCRIPTION:
Deadman Creek 156.0
END DESCRIPTION:
XS GIS Cut Line= 3
      1630905.00      6863237.96      1631005.00      6864838.00
      1631051.89      6865518.02
#Sta/Elev= 30
  3391.3 1825.12  3441.4 1822.88  3491.5 1818.62  3581.7 1813.97  3629.3 1809.69
  3691.9 1806.13  3732.0 1801.18  3794.6 1789.55  3822.2 1783.07  3872.3 1779.41
  4142.8 1775.03  4182.9 1776.49  4323.2 1777.46  4493.5 1776.47  4693.9 1778.10
  4764.0 1777.29  4864.2 1775.13  4894.3 1773.06  4944.4 1772.69  4984.4 1763.90
  4995.0 1763.21  4995.6 1762.71  5022.4 1763.21  5044.6 1769.34  5074.7 1771.04
  5104.7 1777.01  5164.9 1779.83  5555.8 1782.11  5644.8 1784.89  5676.1 1784.63
#Mann=3,-1,0
  3391.3    0.05       0  4995.0    0.05       0  5022.4    0.05       0
Bank Sta=4995,5022.4
Exp/Cntr=0.3,0.1
