HEC-RAS study Deadman Creek.prj: Deadman Creek Base Level Engineering

--- Deadman Creek.g01 (geometry) --- (continued)

Type RM Length L Ch R = 1,129713,578,578,578
BEGIN DESCRIPTION:
Mapping XS e20c4c4d
END DESCRIPTION:
XS GIS Cut Line= 3
      1630582.90      6863599.64      1630497.55      6864962.91
      1630950.36      6865551.05
#Sta/Elev= 30
  3944.3 1808.05  4022.8 1803.45  4072.9 1792.40  4143.0 1782.86  4149.4 1780.65
  4154.4 1781.32  4173.1 1778.35  4203.2 1776.48  4243.2 1776.31  4323.4 1773.14
  4443.6 1776.53  4724.2 1774.69  4834.4 1774.52  4874.5 1775.81  4944.6 1774.36
  4955.3 1773.17  4964.7 1771.66  4974.7 1765.66  4977.5 1762.67  4978.3 1762.17
  5014.1 1762.67  5034.8 1768.14  5064.8 1767.75  5074.9 1768.88  5110.4 1769.10
  5185.1 1776.06  5405.0 1776.44  5555.1 1778.60  5804.3 1779.00  6052.5 1783.24
#Mann=3,-1,0
  3944.3    0.05       0  4977.5    0.03       0  5014.1    0.05       0
Bank Sta=4977.5,5014.1
Exp/Cntr=0.3,0.1

Type RM Length L Ch R = 1,129135,570,570,570
BEGIN DESCRIPTION:
Deadman Creek 155.0
END DESCRIPTION:
XS GIS Cut Line= 3
      1629742.02      6863819.81      1630005.00      6864488.00
      1631104.98      6866037.97
#Sta/Elev= 30
  4281.4 1783.59  4353.6 1782.42  4358.9 1781.03  4451.4 1776.52  4881.6 1773.42
  4978.0 1763.61  4996.8 1766.29  5027.8 1766.95  5078.2 1765.64  5093.0 1763.20
  5099.1 1764.83  5105.4 1762.76  5106.4 1762.26  5151.9 1762.76  5158.2 1766.16
  5164.3 1765.94  5171.1 1770.19  5179.1 1772.75  5185.2 1771.90  5193.9 1774.69
  5207.9 1775.20  5220.9 1772.29  5257.0 1772.01  5342.8 1774.14  5687.1 1776.61
  5931.4 1776.46  6269.0 1778.92  6628.3 1786.40  6771.0 1794.40  6900.1 1799.47
#Mann=3,-1,0
  4281.4    0.05       0  5105.4    0.03       0  5151.9    0.05       0
Bank Sta=5105.4,5151.9
Exp/Cntr=0.3,0.1

Type RM Length L Ch R = 1,128565,536,536,536
BEGIN DESCRIPTION:
Deadman Creek 154.0
END DESCRIPTION:
XS GIS Cut Line= 3
      1629304.98      6864337.96      1629505.00      6864688.00
      1631055.01      6866238.01
#Sta/Elev= 30
  4597.0 1801.37  4735.3 1791.80  4744.6 1790.24  4781.3 1779.01  4825.2 1771.41
  4862.0 1769.54  4905.9 1772.32  4954.8 1772.43  4964.9 1768.94  4970.6 1763.05
  4977.0 1760.29  4977.5 1759.79  5000.2 1760.29  5003.7 1763.97  5014.3 1764.49
  5028.4 1762.84  5056.7 1766.78  5085.0 1767.84  5141.6 1772.72  5622.4 1772.65
  6075.0 1774.36  6357.8 1776.33  6640.6 1780.03  6796.2 1783.39  6824.5 1785.58
  6909.3 1787.50  6994.2 1793.41  7093.2 1798.27  7107.3 1800.07  7192.2 1801.17
#Mann=3,-1,0
  4597.0    0.05       0  4977.0    0.05       0  5000.2    0.05       0
Bank Sta=4977,5000.2
Exp/Cntr=0.3,0.1

Type RM Length L Ch R = 1,128029,546,546,546
BEGIN DESCRIPTION:
Deadman Creek 153.0
END DESCRIPTION:
XS GIS Cut Line= 3
      1628805.03      6865038.00      1629205.00      6865088.00
      1630754.99      6866337.99
#Sta/Elev= 30
  4601.6 1806.14  4762.8 1800.75  4863.6 1791.45  4886.3 1786.68  4903.9 1779.00
  4934.1 1769.74  4961.8 1758.60  4967.5 1758.35  4968.2 1757.85  5000.1 1758.35
  5002.2 1762.56  5007.9 1762.56  5011.9 1764.39  5032.7 1761.55  5055.0 1766.88
  5104.6 1770.01  5168.6 1772.24  5247.0 1769.93  5317.4 1770.02  5395.7 1768.35
  5459.7 1770.27  5622.9 1770.58  5651.6 1771.62  6235.4 1776.37  6334.6 1776.14
  6448.1 1778.28  6555.3 1778.08  6860.8 1782.34  6988.7 1787.86  6995.9 1789.36
#Mann=3,-1,0
  4601.6    0.05       0  4967.5    0.03       0  5000.1    0.05       0
Bank Sta=4967.5,5000.1
Exp/Cntr=0.3,0.1

Type RM Length L Ch R = 1,127483,550,550,550
BEGIN DESCRIPTION:
Deadman Creek 152.0
END DESCRIPTION:
XS GIS Cut Line= 3
      1628805.00      6865388.00      1629155.00      6865588.00
      1630734.20      6866512.86
#Sta/Elev= 30
  4597.8 1800.78  4670.5 1796.19  4751.1 1788.82  4782.1 1784.76  4810.2 1777.44
  4826.0 1771.03  4862.7 1763.86  4912.4 1763.88  4977.9 1760.04  4982.0 1758.07
  4982.5 1757.57  5005.3 1758.07  5024.1 1758.90  5030.2 1762.03  5036.0 1762.75
  5045.9 1766.72  5051.7 1765.74  5067.4 1769.32  5094.7 1770.40  5147.5 1767.42
  5249.2 1767.45  5563.9 1772.22  5915.8 1774.52  6032.3 1776.72  6097.6 1776.30
  6359.5 1780.13  6637.1 1781.49  6717.2 1783.17  6727.1 1784.57  6831.0 1788.00
#Mann=3,-1,0
  4597.8    0.05       0  4982.0    0.05       0  5005.3    0.05       0
Bank Sta=4982,5005.3
Exp/Cntr=0.3,0.1

Type RM Length L Ch R = 1,126933,531,531,531
BEGIN DESCRIPTION:
Deadman Creek 151.0
END DESCRIPTION:
XS GIS Cut Line= 3
      1628754.97      6865737.96      1629005.00      6866088.00
      1630275.86      6867018.06
#Sta/Elev= 30
  4570.6 1791.57  4628.4 1788.37  4670.2 1784.31  4714.4 1782.48  4750.1 1778.60
  4764.8 1775.08  4771.0 1770.73  4806.6 1765.05  4828.7 1763.33  4857.0 1766.31
  4877.9 1766.43  4907.4 1763.46  4943.0 1764.15  4951.6 1763.10  4976.8 1755.84
  4977.7 1755.34  5019.0 1755.84  5029.0 1756.48  5043.6 1763.19  5050.3 1764.40
  5087.5 1767.93  5259.0 1767.64  5516.1 1770.25  5595.6 1772.15  6066.5 1776.19
  6224.9 1780.04  6239.5 1781.34  6260.4 1780.19  6417.1 1786.63  6575.6 1789.92
#Mann=3,-1,0
  4570.6    0.05       0  4976.8    0.03       0  5019.0    0.05       0
Bank Sta=4976.8,5019
Exp/Cntr=0.3,0.1

Type RM Length L Ch R = 1,126402,611,611,611
BEGIN DESCRIPTION:
Deadman Creek 150.0
END DESCRIPTION:
XS GIS Cut Line= 3
      1628605.00      6865738.00      1628705.00      6866438.00
      1629805.03      6867838.04
#Sta/Elev= 30
  4293.7 1796.40  4414.9 1788.20  4445.2 1787.15  4475.5 1784.26  4536.1 1781.54
  4657.4 1772.01  4748.3 1768.52  4829.1 1763.75  4930.1 1761.09  4993.6 1757.11
  4994.3 1756.61  5026.5 1757.11  5051.4 1760.53  5086.6 1762.64  5093.0 1763.99
  5186.1 1766.39  5384.9 1767.65  5407.5 1768.85  5542.2 1768.43  5898.3 1771.15
  6061.8 1774.15  6111.6 1774.13  6247.1 1777.73  6411.6 1787.77  6467.7 1789.46
  6511.0 1792.63  6603.2 1796.89  6616.8 1796.00  6624.9 1797.12  6781.3 1801.56
#Mann=3,-1,0
  4293.7    0.05       0  4993.6    0.03       0  5026.5    0.05       0
Bank Sta=4993.6,5026.5
Exp/Cntr=0.3,0.1

Type RM Length L Ch R = 1,125791,521,521,521
BEGIN DESCRIPTION:
Deadman Creek 149.0
END DESCRIPTION:
XS GIS Cut Line= 3
      1628056.03      6866081.71      1628301.90      6866773.27
      1629208.14      6867820.14
#Sta/Elev= 30
  4189.2 1778.67  4350.0 1767.92  4418.8 1767.92  4499.0 1766.12  4599.2 1766.43
  4858.5 1765.06  4914.9 1763.33  4923.0 1761.43  4970.9 1757.46  4978.5 1754.20
  4985.2 1752.84  4998.9 1752.58  4999.4 1752.08  5022.4 1752.58  5027.9 1754.38
  5035.2 1759.69  5042.2 1761.81  5048.8 1762.26  5063.0 1760.61  5070.7 1760.84
  5127.7 1765.97  5502.8 1766.44  5723.0 1768.11  5928.3 1772.22  5992.0 1772.38
  6069.8 1775.12  6077.5 1774.06  6133.5 1775.73  6198.1 1776.24  6307.8 1780.63
#Mann=3,-1,0
  4189.2    0.05       0  4998.9    0.03       0  5022.4    0.05       0
Bank Sta=4998.9,5022.4
Exp/Cntr=0.3,0.1

Type RM Length L Ch R = 1,125270,540,540,540
BEGIN DESCRIPTION:
Deadman Creek 148.0
END DESCRIPTION:
XS GIS Cut Line= 3
      1627833.15      6865622.27      1627955.00      6867138.00
      1628077.91      6867773.09
#Sta/Elev= 30
  3474.1 1791.70  3600.2 1790.35  3812.6 1785.08  3831.0 1783.35  3891.2 1781.40
  3921.3 1777.84  4021.6 1771.88  4051.7 1768.60  4081.8 1767.04  4914.5 1762.48
  4974.7 1758.14  4992.2 1753.03  5009.6 1750.64  5010.4 1750.14  5047.2 1750.64
  5055.8 1752.59  5072.4 1760.59  5096.6 1764.05  5249.4 1763.46  5284.6 1762.38
  5320.7 1758.31  5336.4 1760.29  5412.3 1765.29  5445.0 1764.56  5491.7 1770.29
  5496.8 1769.60  5543.5 1777.68  5548.6 1776.68  5565.1 1780.47  5641.6 1787.50
#Mann=3,-1,0
  3474.1    0.05       0  5009.6    0.03       0  5047.2    0.05       0
Bank Sta=5009.6,5047.2
Exp/Cntr=0.3,0.1

Type RM Length L Ch R = 1,124730,579,579,579
BEGIN DESCRIPTION:
Deadman Creek 147.0
END DESCRIPTION:
XS GIS Cut Line= 3
      1627385.23      6865851.38      1627505.00      6867338.00
      1627455.01      6867737.95
#Sta/Elev= 30
  3502.6 1785.37  3639.7 1777.81  3690.7 1773.16  3740.0 1770.35  3813.1 1768.63
  3820.2 1766.77  3840.3 1768.08  3850.3 1766.83  3880.4 1766.02  3935.6 1766.51
  4211.5 1762.98  4663.0 1762.63  4823.5 1760.23  4935.3 1761.17  4943.9 1760.77
  4963.9 1756.96  4974.0 1757.12  4984.0 1752.69  4995.3 1751.41  4995.8 1750.91
  5018.9 1751.41  5064.6 1759.01  5112.4 1761.92  5117.5 1760.85  5175.4 1766.36
  5235.9 1770.06  5273.7 1770.45  5326.6 1775.90  5377.0 1778.51  5397.1 1780.66
#Mann=3,-1,0
  3502.6    0.05       0  4995.3    0.05       0  5018.9    0.05       0
Bank Sta=4995.3,5018.9
Exp/Cntr=0.3,0.1

Type RM Length L Ch R = 1,124151,250,250,250
BEGIN DESCRIPTION:
Deadman Creek 146.0
END DESCRIPTION:
XS GIS Cut Line= 3
      1626916.48      6865903.49      1626955.00      6867438.00
      1627061.99      6867824.17
#Sta/Elev= 30
  3465.2 1777.13  3605.1 1769.35  3679.8 1767.25  3689.8 1767.76  3729.8 1765.59
  3939.9 1762.28  4250.0 1759.72  4460.0 1761.28  4710.1 1760.13  4760.1 1760.94
  4780.1 1759.77  4790.1 1757.75  4798.0 1754.72  4803.0 1754.53  4820.1 1757.01
  4850.1 1758.18  4930.2 1756.63  4950.2 1757.47  4970.2 1756.16  4990.2 1751.08
  4993.5 1748.80  4994.0 1748.30  5017.1 1748.80  5017.3 1750.85  5022.5 1751.35
  5041.7 1757.64  5062.4 1762.37  5124.7 1767.26  5176.6 1773.74  5400.9 1783.22
#Mann=3,-1,0
  3465.2    0.05       0  4993.5    0.05       0  5017.1    0.05       0
Bank Sta=4993.5,5017.1
Exp/Cntr=0.3,0.1

Type RM Length L Ch R = 1,123901,373,373,373
BEGIN DESCRIPTION:
Mapping XS c9b0c5d8
END DESCRIPTION:
XS GIS Cut Line= 3
      1626523.07      6866105.62      1626707.19      6867448.39
      1626823.96      6867780.73
#Sta/Elev= 30
  3655.5 1766.99  3678.1 1766.97  3698.3 1765.28  3920.3 1761.48  4182.8 1758.93
  4495.7 1760.14  4778.3 1759.76  4818.7 1760.29  4879.2 1759.53  4909.5 1755.79
  4929.7 1754.14  4956.4 1753.52  4970.1 1755.22  4980.2 1753.38  4988.4 1749.79
  4988.9 1749.29  5012.0 1749.79  5022.8 1749.98  5042.2 1752.49  5063.4 1751.75
  5074.0 1753.72  5079.5 1756.67  5084.8 1757.55  5110.5 1758.53  5148.2 1762.90
  5222.4 1767.60  5234.4 1769.25  5260.1 1770.77  5265.4 1771.94  5363.1 1775.75
#Mann=3,-1,0
  3655.5    0.05       0  4988.4    0.05       0  5012.0    0.05       0
Bank Sta=4988.4,5012
Exp/Cntr=0.3,0.1

Type RM Length L Ch R = 1,123528,215,215,215
BEGIN DESCRIPTION:
Deadman Creek 145.0
END DESCRIPTION:
XS GIS Cut Line= 3
      1625747.24      6866153.17      1626348.83      6867495.86
      1626641.87      6867844.45
#Sta/Elev= 30
  3528.7 1785.23  3560.6 1783.68  3635.7 1777.47  3653.4 1773.81  3687.5 1770.31
  3742.2 1761.01  3917.5 1758.31  4150.0 1759.13  4225.0 1757.95  4607.0 1757.66
  4892.8 1759.36  4947.6 1758.24  4982.2 1755.52  4998.2 1746.69  4998.7 1746.19
  5021.8 1746.69  5034.2 1749.09  5041.9 1753.37  5048.5 1753.84  5083.6 1754.40
  5105.7 1752.83  5147.4 1753.74  5155.1 1754.99  5190.3 1757.40  5225.4 1761.98
  5254.0 1764.38  5276.1 1765.49  5403.6 1768.10  5446.5 1769.51  5455.4 1770.76
#Mann=3,-1,0
  3528.7    0.05       0  4998.2    0.03       0  5021.8    0.05       0
Bank Sta=4998.2,5021.8
Exp/Cntr=0.3,0.1

Type RM Length L Ch R = 1,123313,300,300,300
BEGIN DESCRIPTION:
Mapping XS 7e7b5932
END DESCRIPTION:
XS GIS Cut Line= 3
      1625671.58      6866459.41      1626175.06      6867600.93
      1626308.90      6867924.74
#Sta/Elev= 30
  3714.0 1762.18  3836.1 1758.81  4080.2 1757.32  4277.7 1756.82  4411.9 1757.98
  4428.5 1757.27  4602.7 1757.55  4730.2 1759.54  4739.8 1758.85  4846.8 1758.60
  4860.1 1758.38  4870.1 1756.34  4875.6 1756.19  4881.9 1754.21  4892.8 1753.07
  4927.7 1752.11  4936.6 1749.12  4945.6 1750.38  4969.2 1749.39  4974.6 1750.23
  4987.5 1747.59  4988.0 1747.09  5011.1 1747.59  5012.6 1749.19  5022.4 1752.87
  5057.2 1754.75  5081.1 1754.62  5105.0 1757.35  5182.1 1759.61  5312.0 1761.68
#Mann=3,-1,0
  3714.0    0.05       0  4987.5    0.05       0  5011.1    0.05       0
Bank Sta=4987.5,5011.1
Exp/Cntr=0.3,0.1

Type RM Length L Ch R = 1,123013,262,262,262
BEGIN DESCRIPTION:
Deadman Creek 144.0
END DESCRIPTION:
XS GIS Cut Line= 3
      1625298.35      6866581.01      1625905.00      6867688.00
      1626254.98      6868237.97
#Sta/Elev= 30
  3737.6 1774.38  3800.2 1766.78  3805.9 1765.08  3822.0 1763.88  3827.7 1761.94
  3849.5 1759.33  3865.6 1758.59  4099.8 1756.20  4344.4 1755.37  4681.9 1757.56
  4888.5 1757.58  4942.6 1755.27  4948.3 1755.85  4970.1 1750.50  4977.1 1747.18
  4986.7 1745.28  4987.2 1744.78  5010.4 1745.28  5013.5 1746.12  5035.5 1746.00
  5043.9 1750.04  5049.9 1751.52  5086.3 1751.01  5165.9 1756.85  5383.5 1759.08
  5450.3 1762.08  5462.2 1765.10  5492.7 1767.84  5535.0 1769.34  5651.8 1770.33
#Mann=3,-1,0
  3737.6    0.05       0  4986.7    0.05       0  5010.4    0.05       0
Bank Sta=4986.7,5010.4
Exp/Cntr=0.3,0.1

Type RM Length L Ch R = 1,122751,269,269,269
BEGIN DESCRIPTION:
Mapping XS fe411f91
END DESCRIPTION:
XS GIS Cut Line= 3
      1625068.27      6866854.38      1625715.00      6867839.65
      1626083.62      6868143.22
#Sta/Elev= 30
  3832.1 1774.24  3926.3 1768.05  3941.3 1766.31  3968.4 1761.21  4019.7 1756.32
  4293.9 1754.89  4315.0 1754.15  4324.1 1752.59  4423.5 1755.76  4583.2 1756.59
  4815.3 1756.20  4842.4 1755.68  4865.1 1753.87  4872.6 1752.33  4878.5 1752.82
  4901.0 1750.59  4923.8 1750.16  4944.9 1748.46  4949.2 1746.77  4950.2 1746.27
  4996.5 1746.77  5002.1 1749.60  5006.7 1750.58  5045.2 1752.75  5080.4 1756.06
  5372.3 1758.53  5407.5 1759.79  5436.2 1763.93  5442.7 1765.63  5488.2 1767.93
#Mann=3,-1,0
  3832.1    0.05       0  4949.2    0.05       0  4996.5    0.05       0
Bank Sta=4949.2,4996.5
Exp/Cntr=0.3,0.1

Type RM Length L Ch R = 1,122482,398,398,398
BEGIN DESCRIPTION:
Deadman Creek 143.0
END DESCRIPTION:
XS GIS Cut Line= 3
      1624854.98      6867087.97      1625455.00      6867888.00
      1626155.04      6868238.02
#Sta/Elev= 30
  3998.3 1775.66  4034.8 1771.97  4148.3 1765.11  4241.0 1752.88  4255.6 1752.19
  4484.8 1755.33  4626.5 1755.19  4655.6 1753.59  4661.9 1755.05  4670.2 1752.97
  4676.5 1754.74  4684.8 1752.91  4691.0 1754.55  4698.3 1752.96  4741.0 1754.90
  4870.2 1754.88  4898.3 1753.93  4934.8 1748.17  4955.6 1748.96  4985.8 1744.60
  4986.3 1744.10  5009.5 1744.60  5012.3 1746.33  5034.7 1749.32  5087.8 1754.73
  5512.6 1757.78  5543.4 1758.80  5593.7 1764.97  5632.8 1767.12  5781.0 1769.68
#Mann=3,-1,0
  3998.3    0.05       0  4985.8    0.05       0  5009.5    0.05       0
Bank Sta=4985.8,5009.5
Exp/Cntr=0.3,0.1

Type RM Length L Ch R = 1,122084,179,179,179
BEGIN DESCRIPTION:
Mapping XS cff60a4b
END DESCRIPTION:
XS GIS Cut Line= 5
      1624283.55      6867616.49      1624551.07      6868024.97
      1625391.01      6868036.47      1625704.55      6868030.72
      1626144.04      6868243.29
#Sta/Elev= 30
  3951.7 1767.78  4018.7 1765.87  4054.9 1763.42  4115.4 1755.68  4120.9 1754.21
  4127.3 1750.80  4142.4 1747.18  4156.7 1745.58  4169.5 1745.51  4234.6 1751.08
  4359.5 1752.81  4703.9 1753.87  4753.9 1755.09  4924.0 1755.93  4934.0 1750.22
  4946.3 1740.74  4947.2 1740.24  4988.8 1740.74  4994.0 1743.22  5027.7 1746.00
  5044.0 1748.96  5194.0 1753.60  5454.0 1754.90  5534.0 1756.82  5616.3 1756.34
  5717.8 1758.34  5757.4 1757.08  5830.7 1757.97  5915.5 1766.16  6081.8 1769.59
#Mann=5,-1,0
  3951.7    0.05       0  4115.4    0.12       0  4234.6    0.05       0
  4946.3    0.05       0  4988.8    0.05       0
Bank Sta=4946.3,4988.8
Exp/Cntr=0.3,0.1

Type RM Length L Ch R = 1,121905,999,999,999
BEGIN DESCRIPTION:
Mapping XS 6e8a3132
END DESCRIPTION:
XS GIS Cut Line= 4
      1624208.12      6867689.90      1624551.90      6868174.31
      1625880.02      6868163.89      1626176.87      6868382.62
#Sta/Elev= 30
  3953.3 1765.03  3992.5 1763.68  4078.6 1756.95  4099.5 1753.74  4129.1 1745.99
  4154.9 1745.34  4178.7 1747.32  4257.5 1751.79  4366.5 1754.21  4393.5 1753.09
  4437.8 1754.36  4570.4 1752.94  4900.4 1754.86  4910.4 1754.24  4930.4 1749.25
  4990.4 1745.13  4995.9 1743.35  4996.4 1742.85  5019.6 1743.35  5040.4 1744.51
  5070.4 1749.21  5130.4 1753.47  5340.4 1754.88  5440.4 1752.08  5500.4 1754.79
  5840.4 1757.01  5895.6 1758.51  5924.8 1762.58  5975.0 1766.16  6244.2 1769.03
#Mann=5,-1,0
  3953.3    0.05       0  4154.9    0.12       0  4178.7    0.05       0
  4995.9    0.03       0  5019.6    0.05       0
Bank Sta=4995.9,5019.6
Exp/Cntr=0.3,0.1

Type RM Length L Ch R = 1,120906,561,561,561
BEGIN DESCRIPTION:
Deadman Creek 141.0
END DESCRIPTION:
XS GIS Cut Line= 3
      1623697.72      6867783.67      1624705.00      6868988.00
      1624855.01      6869488.04
#Sta/Elev= 30
  3434.2 1752.95  3499.3 1759.15  3570.2 1759.25  3676.3 1753.90  3747.9 1746.93
  4017.2 1752.21  4571.6 1752.29  4705.6 1746.63  4713.4 1749.30  4719.9 1746.00
  4727.7 1747.95  4734.2 1745.04  4742.0 1748.00  4769.6 1744.37  4826.6 1749.22
  4840.9 1748.55  4855.2 1743.54  4926.0 1744.21  4961.9 1751.27  4968.5 1750.91
  4995.5 1739.98  4996.0 1739.48  5019.2 1739.98  5059.1 1751.77  5092.1 1751.28
  5108.6 1745.77  5130.4 1746.33  5181.7 1752.51  5295.7 1754.24  5526.3 1766.16
#Mann=3,-1,0
  3434.2    0.05       0  4995.5    0.03       0  5019.2    0.05       0
Bank Sta=4995.5,5019.2
Exp/Cntr=0.3,0.1

Type RM Length L Ch R = 1,120345,559,559,559
BEGIN DESCRIPTION:
Deadman Creek 140.0
END DESCRIPTION:
XS GIS Cut Line= 3
      1623369.61      6867830.57      1624155.00      6868938.00
      1624705.01      6869738.02
#Sta/Elev= 30
  3637.9 1756.83  3761.5 1756.43  3805.8 1752.12  3883.3 1751.35  3978.0 1748.12
  3984.2 1748.79  3999.0 1746.69  4034.7 1745.28  4112.9 1746.56  4227.8 1750.25
  4759.3 1749.55  4830.7 1749.70  4851.6 1750.79  4887.3 1749.20  4902.0 1746.86
  4922.9 1740.48  4931.6 1740.75  4937.7 1742.90  4952.5 1743.72  4958.8 1743.61
  4978.7 1739.87  4979.3 1739.37  5007.1 1739.87  5017.9 1742.78  5044.9 1743.84
  5095.7 1748.48  5347.5 1748.09  5728.9 1755.81  5881.2 1768.93  5966.4 1772.67
#Mann=3,-1,0
  3637.9    0.05       0  4978.7    0.03       0  5007.1    0.05       0
Bank Sta=4978.7,5007.1
Exp/Cntr=0.3,0.1

Type RM Length L Ch R = 1,119786,567,567,567
BEGIN DESCRIPTION:
Deadman Creek 139.0
END DESCRIPTION:
XS GIS Cut Line= 3
      1622768.66      6868462.03      1623905.00      6869388.00
      1624155.02      6869888.04
#Sta/Elev= 30
  3535.4 1758.79  3621.8 1757.65  3736.7 1747.68  3870.9 1742.88  3963.6 1745.63
  4062.7 1745.87  4141.0 1748.98  4567.5 1746.61  4895.0 1748.47  4951.0 1745.38
  4958.9 1742.61  4965.3 1742.86  4979.7 1739.86  4985.2 1735.61  4985.7 1735.11
  5008.9 1735.61  5009.6 1737.70  5015.2 1741.06  5054.4 1741.16  5068.3 1743.08
  5166.2 1738.60  5171.7 1740.73  5188.5 1741.56  5194.1 1743.60  5216.5 1745.93
  5314.3 1746.68  5367.4 1748.85  5417.7 1753.16  5484.8 1762.54  5560.3 1767.74
#Mann=3,-1,0
  3535.4    0.05       0  4985.2    0.05       0  5008.9    0.05       0
Bank Sta=4985.2,5008.9
Exp/Cntr=0.3,0.1

Type RM Length L Ch R = 1,119219,576,576,576
BEGIN DESCRIPTION:
Deadman Creek 138.0
END DESCRIPTION:
XS GIS Cut Line= 3
      1622656.09      6868669.13      1623605.00      6869838.00
      1623955.03      6870038.02
#Sta/Elev= 30
  3494.7 1757.90  3634.9 1756.92  3656.9 1752.86  3671.3 1756.37  3706.5 1751.32
  3727.3 1751.79  3763.7 1745.53  3799.1 1744.71  3869.5 1740.53  3919.1 1744.09
  3976.6 1743.87  4061.3 1746.03  4822.1 1745.66  4886.0 1746.47  4893.9 1747.56
  4993.1 1739.68  4997.0 1736.78  5003.1 1736.78  5006.0 1734.38  5007.0 1733.88
  5053.5 1734.38  5067.2 1736.29  5088.8 1741.97  5094.6 1745.77  5103.9 1746.83
  5116.1 1750.44  5175.2 1756.92  5250.0 1761.63  5330.7 1764.43  5403.4 1768.58
#Mann=3,-1,0
  3494.7    0.05       0  5006.0    0.05       0  5053.5    0.05       0
Bank Sta=5006,5053.5
Exp/Cntr=0.3,0.1

Type RM Length L Ch R = 1,118643,563,563,563
BEGIN DESCRIPTION:
Deadman Creek 137.0
END DESCRIPTION:
XS GIS Cut Line= 3
      1622437.32      6868929.53      1623105.00      6870038.00
      1623405.01      6870338.01
#Sta/Elev= 30
  3706.4 1754.96  3944.0 1753.46  3996.5 1751.61  4037.3 1749.18  4081.9 1741.73
  4113.0 1742.06  4118.8 1740.12  4134.3 1739.35  4206.6 1742.32  4235.3 1745.29
  4738.3 1744.19  4781.0 1743.32  4796.5 1741.50  4812.1 1744.02  4854.8 1744.24
  4870.3 1741.96  4883.7 1738.21  4913.0 1737.86  4942.1 1740.46  4971.3 1740.10
  4977.1 1739.01  4986.8 1734.77  4987.6 1733.36  4988.0 1732.86  5006.6 1733.36
  5014.6 1735.95  5057.0 1735.60  5226.7 1754.03  5325.7 1759.16  5424.7 1761.44
#Mann=3,-1,0
  3706.4    0.05       0  4987.6    0.05       0  5006.6    0.05       0
Bank Sta=4987.6,5006.6
Exp/Cntr=0.3,0.1

Type RM Length L Ch R = 1,118080,595,595,595
BEGIN DESCRIPTION:
Deadman Creek 136.0
END DESCRIPTION:
XS GIS Cut Line= 3
      1622140.45      6869257.67      1622605.00      6870238.00
      1623104.99      6870687.99
#Sta/Elev= 30
  3919.9 1751.25  4042.0 1749.32  4104.3 1749.77  4132.5 1747.94  4185.9 1746.47
  4252.2 1741.12  4274.5 1740.21  4382.7 1741.01  4479.2 1743.48  4570.2 1744.03
  4712.1 1743.54  4803.1 1743.26  4883.0 1744.06  4899.6 1742.47  4905.2 1742.98
  4916.2 1741.98  4927.9 1740.59  4945.1 1736.05  4967.9 1735.29  4989.1 1731.90
  4989.6 1731.40  5012.9 1731.90  5018.6 1735.16  5040.2 1736.14  5047.0 1737.89
  5068.6 1741.06  5114.1 1741.11  5273.8 1743.10  5408.3 1750.34  5677.4 1757.40
#Mann=5,-1,0
  3919.9    0.05       0  4712.1    0.12       0  4989.1    0.07       0
  5012.9    0.12       0  5114.1    0.05       0
Bank Sta=4989.1,5012.9
Exp/Cntr=0.3,0.1

Type RM Length L Ch R = 1,117485,454,454,454
BEGIN DESCRIPTION:
Deadman Creek 135.0
END DESCRIPTION:
XS GIS Cut Line= 4
      1621014.32      6869521.55      1621426.90      6869872.22
      1622288.70      6870604.70      1623054.99      6871138.00
#Sta/Elev= 30
  3327.5 1746.50  3552.0 1745.45  3609.1 1746.81  3687.1 1744.75  3921.0 1742.95
  4219.8 1743.35  4431.7 1738.01  4488.8 1740.80  4722.8 1741.97  4737.0 1741.25
  4772.2 1735.72  4800.7 1738.10  4843.6 1734.19  4907.3 1736.17  4956.7 1734.82
  4985.3 1732.96  4989.9 1731.50  4990.3 1731.00  5009.0 1731.50  5014.1 1735.11
  5020.2 1734.74  5029.0 1739.08  5049.9 1735.16  5064.8 1737.67  5151.2 1743.66
  5172.1 1746.94  5279.5 1751.10  5386.8 1752.26  5553.5 1748.32  5933.6 1759.49
#Mann=3,-1,0
  3327.5    0.05       0  4989.9    0.03       0  5009.0    0.05       0
Bank Sta=4989.9,5009
Exp/Cntr=0.3,0.1

Type RM Length L Ch R = 1,117031,437,437,437
BEGIN DESCRIPTION:
Deadman Creek 134.0
END DESCRIPTION:
XS GIS Cut Line= 4
      1620886.90      6869717.20      1621270.65      6870137.85
      1621955.00      6870888.00      1622454.98      6871287.99
#Sta/Elev= 30
  3409.4 1746.24  3720.3 1743.25  3883.1 1742.81  3932.5 1743.56  3939.2 1742.75
  3978.3 1742.03  4272.3 1741.04  4491.9 1740.92  4541.2 1741.68  4618.9 1735.38
  4640.5 1738.14  4689.8 1738.17  4710.8 1739.25  4810.1 1740.29  4866.9 1740.29
  4887.8 1738.68  4909.4 1739.99  4930.4 1736.11  4944.6 1732.34  4994.2 1731.42
  4995.0 1730.47  4995.4 1729.97  5014.1 1730.47  5030.2 1734.24  5122.3 1745.43
  5243.1 1751.06  5271.9 1753.06  5364.8 1753.71  5406.4 1754.93  5634.5 1756.57
#Mann=3,-1,0
  3409.4    0.05       0  4995.0    0.05       0  5014.1    0.05       0
Bank Sta=4995,5014.1
Exp/Cntr=0.3,0.1

Type RM Length L Ch R = 1,116594,398,398,398
BEGIN DESCRIPTION:
Deadman Creek 133.0
END DESCRIPTION:
XS GIS Cut Line= 5
      1620602.62      6870103.94      1621090.12      6870736.50
      1621458.08      6870841.91      1621643.26      6871151.11
      1622005.03      6871338.02
#Sta/Elev= 30
  3458.2 1743.08  4105.0 1740.33  4233.5 1740.44  4279.0 1741.80  4312.7 1741.02
  4317.9 1739.93  4490.7 1739.40  4679.0 1739.36  4716.0 1739.76  4721.8 1740.51
  4817.1 1734.92  4881.3 1738.41  4933.8 1739.31  4955.1 1738.34  4976.5 1731.75
  4984.7 1729.81  4992.1 1729.27  4996.0 1726.96  4996.5 1726.46  5019.9 1726.96
  5028.0 1730.06  5035.7 1731.72  5111.0 1734.73  5116.6 1733.84  5148.3 1736.41
  5170.8 1739.50  5215.8 1741.44  5294.6 1747.56  5349.0 1749.80  5407.2 1750.92
#Mann=3,-1,0
  3458.2    0.05       0  4996.0    0.03       0  5019.9    0.05       0
Bank Sta=4996,5019.9
Exp/Cntr=0.3,0.1

Type RM Length L Ch R = 1,116196,184,184,184
BEGIN DESCRIPTION:
Mapping XS b73a0971
END DESCRIPTION:
XS GIS Cut Line= 5
      1620531.86      6870449.69      1620876.73      6870809.29
      1621300.75      6871295.34      1621415.33      6871486.31
      1621949.82      6871840.04
#Sta/Elev= 30
  3855.8 1741.98  4231.6 1740.48  4281.3 1742.10  4295.4 1740.74  4323.7 1739.87
  4657.1 1737.87  4812.8 1737.91  4876.4 1739.13  4933.3 1730.86  4954.2 1729.96
  4968.4 1730.39  4982.1 1726.05  4982.8 1725.55  5017.0 1726.05  5018.3 1726.26
  5025.5 1731.16  5033.9 1733.67  5055.3 1737.23  5107.1 1739.55  5208.8 1739.54
  5302.8 1737.90  5417.1 1738.05  5453.3 1734.01  5483.4 1736.94  5597.7 1741.84
  5641.1 1745.51  5721.1 1747.06  5778.2 1747.08  5785.0 1747.75  5862.7 1747.49
#Mann=3,-1,0
  3855.8    0.05       0  4982.1    0.03       0  5017.0    0.05       0
Bank Sta=4982.1,5017
Exp/Cntr=0.3,0.1

Type RM Length L Ch R = 1,116012,278,278,278
BEGIN DESCRIPTION:
Mapping XS 7066595c
END DESCRIPTION:
XS GIS Cut Line= 5
      1620401.44      6870823.11      1621102.61      6871301.63
      1621138.39      6871360.02      1621322.52      6871616.01
      1621849.16      6871912.98
#Sta/Elev= 30
  4085.7 1739.90  4623.2 1739.07  4847.5 1737.09  4919.3 1738.17  4933.0 1736.53
  4954.2 1729.46  4977.2 1728.03  4984.0 1726.18  4984.4 1725.68  5004.0 1726.18
  5006.3 1729.16  5027.2 1729.99  5062.8 1736.12  5092.2 1738.34  5113.1 1737.79
  5163.4 1739.01  5234.6 1738.15  5278.8 1739.11  5308.2 1738.18  5344.2 1739.21
  5454.0 1738.13  5475.7 1736.94  5550.9 1737.75  5578.3 1734.12  5599.9 1733.36
  5637.5 1737.34  5711.6 1739.34  5777.6 1743.12  5858.5 1744.24  5923.0 1743.62
#Mann=3,-1,0
  4085.7    0.05       0  4984.0    0.03       0  5004.0    0.05       0
Bank Sta=4984,5004
Exp/Cntr=0.3,0.1

Type RM Length L Ch R = 1,115734,244,244,244
BEGIN DESCRIPTION:
Mapping XS b342220d
END DESCRIPTION:
XS GIS Cut Line= 3
      1620217.74      6871063.62      1621223.72      6871719.30
      1621856.82      6872131.94
#Sta/Elev= 30
  4159.9 1738.80  4681.8 1738.68  4776.4 1738.00  4833.7 1734.75  4860.9 1734.41
  4869.9 1734.89  4875.9 1739.50  4884.8 1741.00  4906.1 1735.91  4942.4 1734.89
  4972.2 1726.29  4972.8 1725.79  5002.2 1726.29  5005.6 1727.89  5051.0 1730.77
  5072.1 1736.00  5087.2 1737.66  5259.2 1738.49  5398.0 1737.70  5425.1 1738.64
  5600.3 1736.26  5648.7 1737.33  5678.7 1733.06  5693.8 1732.92  5708.4 1733.55
  5714.9 1735.25  5720.9 1734.93  5736.0 1736.93  5968.4 1737.66  6116.4 1744.05
#Mann=3,-1,0
  4159.9    0.05       0  4972.2    0.03       0  5002.2    0.05       0
Bank Sta=4972.2,5002.2
Exp/Cntr=0.3,0.1

Type RM Length L Ch R = 1,115490,743,743,743
BEGIN DESCRIPTION:
Deadman Creek 132.0
END DESCRIPTION:
XS GIS Cut Line= 4
      1619488.07      6870878.45      1620833.01      6871737.26
      1621169.83      6871930.37      1621783.86      6872282.42
#Sta/Elev= 30
  3437.9 1739.63  3782.5 1738.13  3897.6 1739.04  3906.9 1737.94  4043.8 1738.91
  4147.2 1738.93  4159.2 1739.05  4337.2 1737.83  4855.3 1736.33  4897.6 1736.41
  4928.1 1738.09  4934.0 1737.86  4941.1 1735.51  4970.4 1733.75  4979.9 1724.49
  4980.5 1723.99  5009.9 1724.49  5027.9 1726.81  5043.5 1731.31  5049.2 1730.71
  5070.8 1734.32  5102.4 1736.92  5226.1 1735.43  5344.1 1737.48  5511.0 1737.05
  5600.8 1735.24  5666.3 1731.95  5768.4 1736.48  5935.3 1738.27  6129.7 1746.42
#Mann=7,-1,0
  3437.9    0.05       0  4043.8   0.075       0  4147.2    0.05       0
  4159.2   0.075       0  4337.2    0.05       0  4979.9    0.03       0
  5009.9    0.05       0
Bank Sta=4979.9,5009.9
Exp/Cntr=0.3,0.1

Type RM Length L Ch R = 1,114747,559,559,559
BEGIN DESCRIPTION:
Deadman Creek 131.0
END DESCRIPTION:
XS GIS Cut Line= 4
      1619579.95      6871962.98      1620655.00      6872338.00
      1621225.47      6872429.27      1621677.71      6872501.63
#Sta/Elev= 30
  3870.2 1738.87  4034.4 1737.83  4087.7 1738.68  4175.6 1736.55  4225.0 1737.74
  4246.2 1736.74  4341.5 1736.71  4458.0 1738.38  4669.9 1737.69  4765.2 1736.21
  4837.9 1732.72  4874.3 1732.20  4913.5 1729.15  4924.1 1727.13  4931.1 1724.19
  4955.8 1723.86  4962.2 1722.02  4980.9 1721.00  4981.5 1720.50  5011.0 1721.00
  5029.0 1726.66  5042.3 1734.21  5049.3 1734.97  5140.4 1735.41  5150.6 1736.40
  5241.7 1734.44  5636.7 1735.44  5768.3 1734.38  5970.9 1738.85  6044.5 1743.72
#Mann=3,-1,0
  3870.2    0.05       0  4980.9    0.05       0  5011.0    0.05       0
Bank Sta=4980.9,5011
Exp/Cntr=0.3,0.1

Type RM Length L Ch R = 1,114188,576,576,576
BEGIN DESCRIPTION:
Deadman Creek 130.0
END DESCRIPTION:
XS GIS Cut Line= 3
      1619629.98      6872713.00      1620405.00      6872788.00
      1621792.96      6872973.19
#Sta/Elev= 30
  4221.8 1737.05  4350.7 1735.56  4449.9 1735.04  4839.7 1733.06  4930.1 1733.64
  4940.2 1730.06  4946.9 1726.19  4980.3 1723.15  4991.8 1720.24  4992.1 1719.74
  5006.9 1720.24  5042.0 1725.58  5050.9 1728.00  5081.1 1727.86  5131.6 1725.37
  5141.7 1726.11  5161.9 1730.63  5171.9 1731.55  5182.0 1730.82  5193.3 1726.23
  5202.2 1728.19  5282.9 1734.17  5866.5 1734.72  6095.9 1741.46  6110.2 1738.54
  6130.4 1742.19  6169.0 1741.11  6261.5 1742.87  6362.4 1748.20  6400.7 1748.82
#Mann=5,-1,0
  4221.8    0.05       0  4350.7    0.12       0  4449.9    0.05       0
  4991.8    0.03       0  5006.9    0.05       0
Bank Sta=4991.8,5006.9
Exp/Cntr=0.3,0.1

Type RM Length L Ch R = 1,113612,390,390,390
BEGIN DESCRIPTION:
Mapping XS 2c884942
END DESCRIPTION:
XS GIS Cut Line= 2
      1619779.90      6873298.09      1621274.29      6873323.12
#Sta/Elev= 30
  4225.1 1735.33  4370.2 1735.35  4390.2 1734.30  4410.2 1735.38  4500.2 1735.48
  4580.2 1735.20  4600.2 1734.19  4660.3 1734.68  4690.3 1737.68  4790.3 1739.46
  4820.3 1737.30  4850.3 1733.52  4870.3 1729.14  4880.3 1728.27  4900.3 1728.49
  4910.3 1727.07  4920.3 1723.76  4960.3 1723.37  4997.1 1719.49  4997.7 1718.99
  5027.3 1719.49  5030.3 1723.61  5040.3 1725.94  5070.3 1731.20  5080.3 1731.54
  5320.3 1732.76  5570.4 1736.94  5590.4 1738.36  5630.4 1737.91  5719.7 1739.50
#Mann=3,-1,0
  4225.1    0.05       0  4997.1    0.05       0  5027.3    0.05       0
Bank Sta=4997.1,5027.3
Exp/Cntr=0.3,0.1

Type RM Length L Ch R = 1,113222,626,626,626
BEGIN DESCRIPTION:
Mapping XS f4df6c46
END DESCRIPTION:
XS GIS Cut Line= 2
      1620113.04      6873670.83      1621120.30      6873709.23
#Sta/Elev= 30
  4606.8 1735.88  4720.7 1733.43  4788.9 1731.61  4828.9 1731.90  4909.0 1728.29
  4925.2 1725.69  4949.0 1724.10  4959.0 1719.49  4969.0 1719.05  4979.0 1719.84
  4990.3 1718.80  4990.9 1718.30  5020.6 1718.80  5029.1 1723.06  5039.1 1725.37
  5069.1 1727.07  5109.1 1727.23  5129.1 1726.06  5149.2 1725.89  5169.2 1726.60
  5186.5 1728.46  5191.5 1730.22  5199.2 1731.54  5209.2 1731.96  5269.2 1732.14
  5429.4 1734.82  5469.4 1736.66  5509.4 1736.91  5559.5 1738.97  5614.8 1739.76
#Mann=4,-1,0
  4606.8     0.1       0  4720.7    0.05       0  4990.3    0.05       0
  5020.6    0.05       0
Bank Sta=4990.3,5020.6
Exp/Cntr=0.3,0.1

Type RM Length L Ch R = 1,112596,647,647,647
BEGIN DESCRIPTION:
Mapping XS e4c1d31a
END DESCRIPTION:
XS GIS Cut Line= 2
      1620039.06      6873858.81      1620916.80      6874492.19
#Sta/Elev= 30
  4430.6 1731.96  4508.0 1731.80  4721.6 1729.06  4778.3 1729.57  4857.2 1727.38
  4878.9 1725.33  4885.1 1725.95  4899.8 1725.19  4906.5 1723.81  4929.2 1722.97
  4950.1 1726.12  4970.9 1720.31  4979.5 1719.71  4985.7 1717.20  4987.6 1715.55
  4988.1 1715.05  5012.8 1715.55  5015.1 1718.38  5021.2 1720.46  5035.9 1723.26
  5042.2 1725.52  5092.4 1734.50  5142.7 1735.92  5165.5 1734.82  5207.7 1737.66
  5251.8 1738.31  5264.2 1739.76  5323.0 1739.47  5387.5 1742.34  5513.0 1742.80
#Mann=4,-1,0
  4430.6   0.075       0  4508.0    0.05       0  4987.6    0.05       0
  5012.8    0.05       0
Bank Sta=4987.6,5012.8
Exp/Cntr=0.3,0.1

Type RM Length L Ch R = 1,111949,547,547,547
BEGIN DESCRIPTION:
Deadman Creek 129.0
END DESCRIPTION:
XS GIS Cut Line= 3
      1619350.97      6874315.07      1620055.00      6874638.00
      1620760.57      6874894.20
#Sta/Elev= 30
  4220.3 1729.10  4722.2 1728.43  4842.6 1728.63  4860.1 1729.49  4873.8 1728.25
  4883.1 1728.86  4906.1 1728.35  4917.8 1729.58  4934.6 1727.85  4950.8 1727.70
  4972.9 1728.85  4986.1 1726.59  4992.1 1721.56  4994.5 1712.97  4995.1 1712.47
  5024.8 1712.97  5026.8 1713.22  5035.4 1717.55  5058.7 1718.23  5080.0 1720.36
  5090.6 1720.65  5096.7 1722.81  5111.9 1725.19  5165.1 1724.77  5213.8 1726.78
  5244.4 1726.73  5324.7 1729.47  5392.1 1730.21  5539.8 1736.96  5745.5 1737.09
#Mann=3,-1,0
  4220.3    0.05       0  4994.5    0.03       0  5024.8    0.05       0
Bank Sta=4994.5,5024.8
Exp/Cntr=0.3,0.1

Type RM Length L Ch R = 1,111402,531,531,531
BEGIN DESCRIPTION:
Deadman Creek 128.0
END DESCRIPTION:
XS GIS Cut Line= 3
      1618530.00      6874913.00      1619805.00      6875088.00
      1620691.94      6875074.08
#Sta/Elev= 30
  3708.4 1732.15  4367.4 1730.69  4430.1 1731.17  4722.8 1727.25  4914.6 1727.28
  4924.7 1728.19  4934.8 1728.07  4959.3 1726.67  4975.2 1724.84  4985.3 1722.62
  4992.8 1718.91  4997.9 1718.91  5005.4 1715.03  5020.1 1711.77  5021.1 1711.27
  5070.6 1711.77  5085.4 1717.49  5095.4 1722.46  5105.4 1724.39  5115.4 1724.66
  5125.4 1723.81  5145.4 1725.84  5175.4 1724.79  5312.2 1724.78  5455.4 1727.47
  5605.4 1727.89  5745.4 1729.79  5775.5 1731.78  5815.5 1731.71  5882.4 1735.61
#Mann=3,-1,0
  3708.4    0.05       0  5020.1    0.03       0  5070.6    0.05       0
Bank Sta=5020.1,5070.6
Exp/Cntr=0.3,0.1

Type RM Length L Ch R = 1,110871,424,424,424
BEGIN DESCRIPTION:
Deadman Creek 127.0
END DESCRIPTION:
XS GIS Cut Line= 3
      1618580.02      6875813.00      1620005.00      6875538.00
      1621254.98      6874838.01
#Sta/Elev= 30
  3550.0 1729.05  4555.5 1728.54  4756.8 1724.39  4807.8 1717.93  4828.1 1717.67
  4848.5 1719.61  4871.6 1719.90  4899.4 1716.61  4950.3 1716.34  4956.0 1714.62
  4956.8 1714.12  4996.4 1714.62  4998.7 1719.83  5009.3 1720.35  5024.2 1724.20
  5052.6 1725.92  5112.0 1724.49  5310.7 1726.83  5604.0 1727.38  5641.7 1728.35
  5793.5 1736.48  5852.9 1735.61  5906.5 1737.92  5933.9 1737.09  6015.0 1738.24
  6036.7 1739.78  6117.7 1739.48  6177.1 1741.99  6227.6 1741.76  6433.9 1746.21
#Mann=3,-1,0
  3550.0    0.05       0  4956.0    0.05       0  4996.4    0.05       0
Bank Sta=4956,4996.4
Exp/Cntr=0.3,0.1

Type RM Length L Ch R = 1,110447,527,527,527
BEGIN DESCRIPTION:
Mapping XS 8f64d95a
END DESCRIPTION:
XS GIS Cut Line= 2
      1619515.15      6876091.60      1620965.90      6875650.95
#Sta/Elev= 30
  4287.3 1728.55  4730.5 1728.06  4778.3 1725.64  4788.8 1726.11  4841.1 1722.44
  4893.3 1721.20  4945.6 1713.73  4966.1 1707.77  4966.8 1707.27  5001.5 1707.77
  5004.0 1715.40  5009.3 1714.49  5018.7 1716.37  5036.9 1722.12  5042.2 1720.59
  5050.1 1722.27  5069.8 1723.36  5227.7 1724.38  5315.6 1723.88  5321.8 1721.19
  5332.3 1721.23  5348.5 1724.78  5386.6 1726.93  5414.3 1729.76  5490.5 1730.32
  5530.8 1733.91  5666.7 1736.17  5687.6 1735.53  5750.3 1737.64  5803.5 1737.33
#Mann=3,-1,0
  4287.3    0.05       0  4966.1    0.05       0  5001.5    0.05       0
Bank Sta=4966.1,5001.5
Exp/Cntr=0.3,0.1

Type RM Length L Ch R = 1,109920,326,326,326
BEGIN DESCRIPTION:
Mapping XS 997b0aa1
END DESCRIPTION:
XS GIS Cut Line= 2
      1619433.87      6876315.29      1620801.61      6876328.84
#Sta/Elev= 30
  3992.1 1726.83  4153.2 1726.45  4203.2 1727.05  4263.2 1725.74  4463.3 1724.42
  4693.3 1723.87  4703.3 1723.32  4723.3 1723.79  4743.3 1722.70  4763.3 1722.85
  4769.4 1722.17  4793.3 1722.72  4813.3 1722.03  4833.3 1722.68  4863.3 1720.56
  4913.3 1719.83  4933.3 1718.60  4963.3 1714.07  4973.3 1711.66  4974.7 1710.17
  4975.3 1709.67  5004.6 1709.67  5005.2 1710.17  5043.3 1719.51  5053.3 1721.02
  5063.3 1721.43  5093.3 1726.09  5163.3 1731.70  5183.3 1732.24  5359.9 1732.64
#Mann=3,-1,0
  3992.1    0.05       0  4974.7    0.05       0  5005.2    0.05       0
Bank Sta=4974.7,5005.2
Exp/Cntr=0.3,0.1

Type RM Length L Ch R = 1,109594,369,369,369
BEGIN DESCRIPTION:
Mapping XS c8ea93c5
END DESCRIPTION:
XS GIS Cut Line= 3
      1619581.44      6876652.65      1620219.08      6876614.14
      1620720.32      6876663.81
#Sta/Elev= 30
  4173.9 1725.61  4197.5 1725.92  4257.6 1723.93  4598.2 1723.24  4618.3 1722.43
  4658.3 1722.34  4738.5 1723.44  4758.5 1723.28  4778.6 1721.92  4788.6 1722.76
  4818.7 1722.63  4828.7 1722.44  4848.8 1716.11  4919.1 1716.90  4949.3 1716.18
  4989.5 1712.98  4996.0 1710.37  4996.7 1709.87  5030.8 1709.87  5031.5 1710.37
  5039.7 1715.85  5049.8 1717.23  5069.9 1719.56  5100.0 1720.01  5120.1 1721.52
  5140.2 1725.23  5170.4 1727.54  5211.2 1728.48  5230.7 1727.86  5316.4 1728.07
#Mann=3,-1,0
  4173.9    0.05       0  4996.0    0.05       0  5031.5    0.05       0
Bank Sta=4996,5031.5
Exp/Cntr=0.3,0.1

Type RM Length L Ch R = 1,109225,351,351,351
BEGIN DESCRIPTION:
Mapping XS be03128e
END DESCRIPTION:
XS GIS Cut Line= 3
      1619622.31      6876989.44      1620229.54      6876969.78
      1620898.18      6876972.87
#Sta/Elev= 30
  4317.4 1725.48  4400.1 1724.87  4450.2 1725.38  4550.2 1722.71  4700.3 1721.28
  4820.4 1721.17  4870.4 1722.23  4890.4 1721.18  4900.4 1722.62  4910.4 1722.63
  4920.2 1721.13  4940.4 1720.93  4950.4 1719.19  4980.4 1711.26  4982.6 1705.89
  4983.3 1705.39  5017.4 1705.39  5018.1 1705.89  5030.4 1713.37  5040.4 1715.28
  5080.4 1714.78  5100.4 1712.26  5120.4 1712.07  5140.4 1717.50  5150.4 1718.83
  5190.4 1720.50  5220.4 1723.12  5260.4 1723.06  5410.4 1726.93  5593.6 1727.07
#Mann=3,-1,0
  4317.4    0.05       0  4982.6    0.05       0  5018.1    0.05       0
Bank Sta=4982.6,5018.1
Exp/Cntr=0.3,0.1

Type RM Length L Ch R = 1,108874,583,583,583
BEGIN DESCRIPTION:
Mapping XS 6030443e
END DESCRIPTION:
XS GIS Cut Line= 4
      1619571.24      6877285.08      1620260.16      6877320.30
      1620545.62      6877277.93      1620775.00      6877041.80
#Sta/Elev= 30
  4213.7 1726.11  4267.5 1725.25  4337.6 1725.50  4427.7 1724.48  4598.0 1719.12
  4628.0 1718.87  4698.1 1718.75  4888.3 1721.48  4908.5 1721.06  4918.5 1722.42
  4928.6 1722.54  4938.7 1720.99  4953.6 1720.28  4959.0 1718.18  4979.2 1714.83
  4989.3 1712.33  4990.5 1706.61  4991.1 1706.11  5020.3 1706.11  5020.9 1706.61
  5029.7 1706.94  5039.8 1710.81  5100.5 1716.28  5130.8 1719.93  5151.0 1721.05
  5156.8 1721.89  5212.8 1721.42  5354.3 1724.73  5467.5 1726.63  5521.3 1726.96
#Mann=3,-1,0
  4213.7    0.05       0  4990.5    0.03       0  5020.9    0.05       0
Bank Sta=4990.5,5020.9
Exp/Cntr=0.3,0.1

Type RM Length L Ch R = 1,108291,504,504,504
BEGIN DESCRIPTION:
Mapping XS 326ada1b
END DESCRIPTION:
XS GIS Cut Line= 4
      1619500.28      6877705.91      1620321.46      6877821.12
      1621003.66      6877916.83      1621304.89      6878260.90
#Sta/Elev= 30
  4035.1 1724.19  4080.3 1724.39  4201.4 1722.36  4423.6 1716.87  4575.1 1719.05
  4804.1 1720.63  4857.8 1721.89  4863.6 1720.45  4868.6 1720.45  4875.4 1721.76
  4888.1 1721.78  4968.9 1716.03  4979.0 1713.63  4993.4 1705.00  4994.3 1704.30
  5031.1 1704.30  5031.9 1705.00  5059.8 1707.75  5069.9 1710.41  5100.1 1714.84
  5110.2 1715.08  5150.6 1719.22  5160.7 1718.86  5180.9 1719.94  5384.8 1718.87
  5483.9 1720.04  5527.5 1721.42  5654.2 1722.50  5767.4 1721.86  6010.5 1723.80
#Mann=3,-1,0
  4035.1    0.05       0  4993.4    0.03       0  5031.9    0.05       0
Bank Sta=4993.4,5031.9
Exp/Cntr=0.3,0.1

Type RM Length L Ch R = 1,107787,381,381,381
BEGIN DESCRIPTION:
Mapping XS ed2f9eb1
END DESCRIPTION:
XS GIS Cut Line= 3
      1619445.39      6878201.90      1620154.87      6878276.11
      1621228.26      6878388.39
#Sta/Elev= 30
  3934.2 1719.67  4004.2 1719.64  4084.6 1717.65  4236.8 1715.78  4506.9 1718.12
  4738.2 1718.14  4778.4 1718.55  4788.4 1719.61  4806.7 1717.61  4828.7 1718.74
  4858.8 1716.00  4899.0 1714.42  4919.2 1711.39  4939.3 1712.40  4949.3 1711.42
  4969.4 1706.73  4983.1 1705.33  4984.0 1704.63  5020.8 1704.63  5021.6 1705.33
  5029.8 1716.40  5039.8 1718.97  5059.9 1719.92  5361.6 1718.99  5452.0 1717.63
  5485.0 1718.32  5492.3 1719.22  5532.5 1719.19  5643.1 1723.02  5726.8 1723.28
#Mann=3,-1,0
  3934.2    0.05       0  4983.1    0.05       0  5021.6    0.05       0
Bank Sta=4983.1,5021.6
Exp/Cntr=0.3,0.1

Type RM Length L Ch R = 1,107406,132,132,132
BEGIN DESCRIPTION:
Mapping XS 6fc512a6
END DESCRIPTION:
XS GIS Cut Line= 4
      1618993.50      6877978.81      1619299.19      6878669.75
      1619858.82      6878660.79      1621171.63      6878630.84
#Sta/Elev= 30
  3185.4 1721.66  3351.9 1720.76  3611.0 1716.76  3928.1 1714.70  4266.8 1715.07
  4626.9 1718.25  4847.0 1717.89  4866.9 1718.54  4886.9 1715.93  4916.9 1716.63
  4956.9 1713.97  4966.9 1712.32  4977.0 1708.29  4992.7 1706.27  4993.5 1705.57
  5030.3 1705.57  5031.2 1706.27  5037.0 1709.49  5047.0 1710.78  5097.0 1712.51
  5117.0 1711.30  5127.0 1711.74  5137.0 1714.93  5147.0 1716.76  5163.7 1717.51
  5239.2 1717.66  5567.1 1717.87  5627.1 1718.58  5657.1 1721.42  5813.8 1722.17
#Mann=5,-1,0
  3185.4    0.05       0  4992.7    0.05       0  5031.2    0.05       0
  5163.7    0.12       0  5239.2    0.05       0
Bank Sta=4992.7,5031.2
Exp/Cntr=0.3,0.1

Type RM Length L Ch R = 1,107274,324,324,324
BEGIN DESCRIPTION:
Mapping XS 1e5d38c1
END DESCRIPTION:
XS GIS Cut Line= 5
      1618822.01      6877982.21      1619217.60      6878750.07
      1619298.35      6878752.31      1619880.00      6878763.00
      1621321.58      6878770.73
#Sta/Elev= 30
  3049.2 1720.17  3828.6 1715.31  3856.4 1714.00  3865.7 1715.60  3909.0 1712.17
  4300.5 1717.08  4810.5 1718.45  4850.5 1716.63  4900.5 1717.54  4930.5 1710.92
  4950.5 1710.36  4960.5 1708.46  4980.5 1708.52  4989.8 1706.18  4990.5 1705.48
  5022.8 1706.18  5060.5 1711.96  5110.5 1712.58  5140.5 1709.09  5160.5 1714.38
  5172.7 1715.72  5310.5 1716.68  5410.5 1716.17  5440.5 1714.20  5470.8 1715.21
  5560.5 1718.67  5660.5 1719.14  5680.5 1717.38  5700.5 1719.65  6017.1 1723.48
#Mann=5,-1,0
  3049.2    0.05       0  4989.8    0.05       0  5022.8    0.05       0
  5172.7    0.12       0  5470.8    0.05       0
Bank Sta=4989.8,5022.8
Exp/Cntr=0.3,0.1

Type RM Length L Ch R = 1,106950,996,996,996
BEGIN DESCRIPTION:
Mapping XS c4bea2b9
END DESCRIPTION:
XS GIS Cut Line= 5
      1618805.47      6878056.67      1618851.30      6878719.34
      1619124.44      6878777.13      1619768.86      6878910.68
      1620778.44      6879255.54
#Sta/Elev= 30
  2937.6 1720.20  3288.9 1715.62  3520.3 1715.41  3570.4 1716.44  3584.3 1715.32
  3590.5 1716.63  3615.1 1717.10  3620.3 1716.02  3902.0 1711.98  4209.6 1716.69
  4731.3 1717.16  4799.3 1715.53  4919.2 1715.13  4981.8 1710.49  4983.5 1704.26
  4984.2 1703.56  5016.6 1704.26  5031.7 1706.28  5070.5 1707.75  5095.1 1712.40
  5148.0 1716.46  5253.1 1718.11  5264.2 1717.28  5315.7 1718.47  5321.0 1720.03
  5327.6 1720.27  5352.3 1718.91  5401.6 1719.92  5566.3 1726.02  5606.0 1726.42
#Mann=3,-1,0
  2937.6    0.05       0  4983.5    0.05       0  5016.6    0.05       0
Bank Sta=4983.5,5016.6
Exp/Cntr=0.3,0.1

Type RM Length L Ch R = 1,105954,532,532,532
BEGIN DESCRIPTION:
Deadman Creek 126.0
END DESCRIPTION:
XS GIS Cut Line= 5
      1618750.34      6877998.79      1618797.38      6878745.45
      1619403.49      6879056.23      1619802.70      6879791.86
      1620375.25      6880593.43
#Sta/Elev= 30
  3248.8 1719.45  3288.1 1720.18  3338.2 1719.56  3368.2 1717.98  3658.8 1715.36
  3899.3 1715.20  3939.4 1716.14  3949.4 1715.05  3969.4 1716.95  3989.5 1715.56
  4264.0 1711.95  4500.6 1715.60  4819.9 1716.41  4901.7 1715.53  4930.4 1710.89
  4945.4 1709.67  4953.1 1708.27  4961.6 1704.82  4967.2 1705.27  4973.1 1703.11
  4973.9 1702.41  5011.7 1703.11  5021.4 1706.23  5027.1 1706.61  5092.7 1707.35
  5130.8 1712.08  5203.5 1714.19  5872.3 1717.38  5952.1 1716.84  6500.1 1720.47
#Mann=3,-1,0
  3248.8    0.05       0  4973.1    0.05       0  5011.7    0.05       0
Bank Sta=4973.1,5011.7
Exp/Cntr=0.3,0.1

Type RM Length L Ch R = 1,105422,504,504,504
BEGIN DESCRIPTION:
Deadman Creek 125.0
END DESCRIPTION:
XS GIS Cut Line= 4
      1618587.69      6877893.98      1618667.87      6878761.01
      1619105.00      6879538.00      1620072.16      6880724.90
#Sta/Elev= 30
  3236.9 1718.68  3873.6 1715.02  4044.4 1715.36  4064.4 1716.61  4084.5 1715.28
  4287.8 1714.73  4448.4 1711.69  4910.2 1713.81  4963.8 1712.06  4969.5 1709.21
  4991.2 1704.50  4995.2 1700.57  4996.0 1699.87  5033.8 1700.57  5035.1 1704.42
  5049.4 1704.72  5076.7 1707.83  5084.6 1707.20  5091.1 1705.04  5134.1 1702.58
  5177.2 1705.08  5198.1 1712.04  5205.5 1712.01  5218.9 1709.37  5247.6 1709.20
  5311.5 1713.06  5383.3 1714.80  5517.6 1712.91  6044.0 1719.17  6530.2 1718.92
#Mann=3,-1,0
  3236.9    0.05       0  4995.2    0.05       0  5033.8    0.05       0
Bank Sta=4995.2,5033.8
Exp/Cntr=0.3,0.1

Type RM Length L Ch R = 1,104918,611,611,611
BEGIN DESCRIPTION:
Deadman Creek 124.0
END DESCRIPTION:
XS GIS Cut Line= 4
      1618339.60      6877951.93      1618357.79      6878793.52
      1618781.87      6879776.24      1619344.37      6881260.63
#Sta/Elev= 30
  3075.2 1719.25  3511.4 1715.00  3771.4 1714.49  3821.4 1715.78  3831.4 1714.64
  3841.4 1716.29  3861.5 1714.55  4259.5 1714.16  4556.3 1712.58  4679.3 1710.22
  4784.2 1710.46  4836.7 1712.22  4869.4 1708.36  4891.2 1703.14  4923.9 1700.86
  4954.2 1706.27  4959.7 1705.83  4977.7 1702.55  4980.6 1698.89  4981.5 1698.19
  5019.3 1698.89  5021.3 1703.06  5032.0 1704.46  5037.9 1707.31  5043.2 1707.40
  5062.7 1712.80  5074.7 1713.63  5493.6 1713.77  5823.3 1718.34  6574.7 1716.84
#Mann=3,-1,0
  3075.2    0.05       0  4980.6    0.05       0  5019.3    0.05       0
Bank Sta=4980.6,5019.3
Exp/Cntr=0.3,0.1

Type RM Length L Ch R = 1,104307,644,644,644
BEGIN DESCRIPTION:
Deadman Creek 123.0
END DESCRIPTION:
XS GIS Cut Line= 3
      1617869.59      6878718.14      1618305.00      6879988.00
      1619030.02      6881413.03
#Sta/Elev= 30
  3650.4 1714.51  3671.4 1713.57  3766.5 1713.12  4200.0 1712.84  4325.7 1709.72
  4388.3 1709.26  4612.5 1712.80  4820.8 1711.98  4866.0 1713.20  4926.3 1711.95
  4977.2 1704.76  4990.2 1700.79  4995.6 1700.79  4997.1 1697.33  4997.9 1696.63
  5034.9 1696.63  5035.7 1697.33  5037.7 1699.86  5060.2 1702.39  5067.9 1704.80
  5073.5 1707.92  5082.6 1709.46  5105.0 1710.88  5136.7 1709.82  5229.2 1712.01
  5318.2 1711.24  5512.8 1712.34  5690.8 1715.61  5824.3 1716.54  6591.7 1717.09
#Mann=5,-1,0
  3650.4    0.05       0  4926.3    0.12       0  4997.1    0.07       0
  5035.7    0.12       0  5136.7    0.05       0
Bank Sta=4997.1,5035.7
Exp/Cntr=0.3,0.1

Type RM Length L Ch R = 1,103663,536,536,536
BEGIN DESCRIPTION:
Mapping XS d8653cb6
END DESCRIPTION:
XS GIS Cut Line= 3
      1617677.91      6878744.46      1617731.40      6880183.45
      1618369.27      6881244.26
#Sta/Elev= 30
  3247.9 1713.45  3271.5 1712.02  3291.5 1711.86  3741.8 1711.66  3981.9 1708.62
  4142.1 1712.15  4809.9 1710.44  4861.1 1711.51  4882.5 1711.23  4913.5 1709.37
  4939.8 1705.35  4971.8 1698.80  4975.9 1696.86  4976.7 1696.16  5013.7 1696.16
  5014.6 1696.86  5035.9 1704.18  5043.2 1705.63  5051.5 1705.06  5057.3 1705.93
  5066.6 1703.41  5072.8 1705.75  5078.6 1704.90  5088.4 1707.60  5094.2 1706.53
  5101.6 1708.27  5137.0 1710.19  5263.2 1711.03  5311.8 1712.43  5925.7 1712.69
#Mann=5,-1,0
  3247.9    0.05       0  4939.8    0.12       0  4975.9    0.07       0
  5014.6    0.12       0  5078.6    0.05       0
Bank Sta=4975.9,5014.6
Exp/Cntr=0.3,0.1

Type RM Length L Ch R = 1,103127,164,164,164
BEGIN DESCRIPTION:
Deadman Creek 122.0
END DESCRIPTION:
XS GIS Cut Line= 3
      1617439.66      6878722.41      1617476.12      6881342.25
      1617949.60      6881753.29
#Sta/Elev= 30
  2984.2 1714.56  3019.8 1714.84  3039.8 1712.62  3709.9 1709.22  3959.9 1711.52
  4650.0 1710.15  4700.0 1711.38  4847.4 1710.43  4870.0 1709.93  4900.0 1707.35
  4930.0 1706.63  4940.0 1705.85  4948.2 1703.61  4960.0 1700.17  4977.8 1697.04
  4978.8 1696.34  5021.1 1696.34  5022.1 1697.04  5030.0 1698.23  5040.0 1703.67
  5050.0 1707.09  5070.0 1708.83  5110.0 1707.93  5340.0 1709.64  5604.3 1709.11
  5841.2 1710.39  5883.8 1709.50  6110.7 1710.71  6125.0 1712.55  6231.3 1712.05
#Mann=5,-1,0
  2984.2    0.05       0  4847.4    0.12       0  4948.2    0.05       0
  4977.8    0.05       0  5022.1    0.05       0
Bank Sta=4977.8,5022.1
Exp/Cntr=0.3,0.1

Type RM Length L Ch R = 1,102963,1027,1027,1027
BEGIN DESCRIPTION:
Mapping XS 572de538
END DESCRIPTION:
XS GIS Cut Line= 3
      1617288.67      6879090.17      1617309.53      6881333.90
      1617833.84      6881804.12
#Sta/Elev= 30
  3357.7 1714.22  3475.5 1714.48  3575.5 1712.59  3665.5 1708.49  3765.5 1707.13
  3865.5 1709.63  4035.6 1711.56  4605.6 1709.40  4935.6 1709.97  4955.6 1708.40
  4975.6 1702.34  4990.3 1699.21  4991.3 1698.51  5033.6 1698.51  5034.6 1699.21
  5055.6 1700.19  5065.6 1702.68  5095.6 1704.85  5175.6 1706.56  5235.6 1706.31
  5445.6 1709.48  5636.3 1708.86  5672.2 1710.02  5770.9 1710.43  5806.8 1709.51
  6047.5 1709.35  6174.5 1711.66  6231.4 1711.24  6259.8 1712.57  6305.8 1712.00
#Mann=3,-1,0
  3357.7    0.05       0  4990.3    0.05       0  5034.6    0.05       0
Bank Sta=4990.3,5034.6
Exp/Cntr=0.3,0.1
