HEC-RAS study Deadman Creek.prj: Deadman Creek Base Level Engineering

--- Deadman Creek.g01 (geometry) --- (continued)

Type RM Length L Ch R = 1,61236,537,537,537
BEGIN DESCRIPTION:
Deadman Creek 70.0
END DESCRIPTION:
XS GIS Cut Line= 3
      1616605.01      6904388.00      1618805.00      6904626.23
      1619186.95      6904634.91
#Sta/Elev= 30
  2786.5 1679.50  2907.2 1677.20  2983.5 1674.28  3020.8 1673.24  3092.0 1668.32
  3219.0 1657.61  3239.1 1653.14  3259.2 1651.08  3369.9 1646.96  3782.3 1645.56
  4314.7 1646.56  4587.0 1645.10  4691.6 1645.71  4707.7 1646.98  4785.3 1644.69
  4798.2 1646.38  4838.4 1640.14  4880.1 1641.23  4949.1 1638.68  4979.2 1640.40
  4986.6 1634.59  4987.0 1634.09  5009.0 1634.59  5021.9 1637.22  5049.4 1646.64
  5099.4 1645.78  5149.4 1646.91  5199.4 1649.77  5279.4 1656.78  5381.4 1660.11
#Mann=7,-1,0
  2786.5    0.05       0  2983.5    0.12       0  3092.0    0.05       0
  4785.3    0.12       0  4986.6    0.07       0  5009.0    0.12       0
  5021.9    0.05       0
Bank Sta=4986.6,5009
Exp/Cntr=0.3,0.1

Type RM Length L Ch R = 1,60699,565,565,565
BEGIN DESCRIPTION:
Deadman Creek 69.0
END DESCRIPTION:
XS GIS Cut Line= 3
      1617005.02      6904688.00      1618605.00      6905088.00
      1619004.98      6905088.00
#Sta/Elev= 30
  3345.3 1664.47  3368.5 1662.79  3386.5 1660.19  3409.7 1660.47  3487.0 1653.08
  3492.2 1653.24  3528.2 1650.19  3706.1 1645.43  3757.6 1645.66  3816.9 1644.65
  4510.1 1645.52  4819.3 1644.51  4901.8 1645.10  4947.2 1644.42  4963.6 1644.72
  4971.3 1642.89  4976.5 1643.05  4984.2 1639.85  4988.6 1632.51  4989.1 1632.01
  5020.5 1632.51  5024.5 1635.03  5044.5 1636.40  5084.5 1642.41  5129.8 1651.12
  5174.5 1655.53  5234.5 1658.41  5294.5 1662.58  5324.5 1665.49  5394.5 1669.80
#Mann=5,-1,0
  3345.3    0.05       0  4947.2    0.12       0  4988.6    0.07       0
  5020.5    0.12       0  5129.8    0.05       0
Bank Sta=4988.6,5020.5
Exp/Cntr=0.3,0.1

Type RM Length L Ch R = 1,60134,564,564,564
BEGIN DESCRIPTION:
Deadman Creek 68.0
END DESCRIPTION:
XS GIS Cut Line= 3
      1616978.54      6905365.28      1618655.00      6905638.00
      1619054.99      6905588.00
#Sta/Elev= 30
  3301.3 1661.47  3500.3 1651.07  3536.0 1650.15  3561.1 1650.58  3632.1 1647.77
  3672.6 1647.86  3720.6 1645.97  3843.7 1643.85  4746.5 1643.99  4858.0 1643.75
  4887.3 1642.25  4910.0 1642.58  4928.9 1641.83  4971.6 1637.43  4979.5 1634.90
  4994.5 1632.17  4995.0 1631.67  5023.2 1632.17  5030.0 1639.81  5037.6 1642.56
  5042.6 1642.38  5050.2 1646.33  5080.4 1650.91  5123.3 1653.86  5147.1 1656.79
  5181.2 1658.96  5211.4 1662.20  5279.5 1666.67  5352.5 1669.26  5402.9 1672.62
#Mann=5,-1,0
  3301.3    0.05       0  4887.3    0.12       0  4994.5    0.07       0
  5023.2    0.12       0  5147.1    0.05       0
Bank Sta=4994.5,5023.2
Exp/Cntr=0.3,0.1

Type RM Length L Ch R = 1,59570,582,582,582
BEGIN DESCRIPTION:
Deadman Creek 67.0
END DESCRIPTION:
XS GIS Cut Line= 3
      1616798.03      6905865.28      1618605.00      6906188.00
      1619005.03      6906087.99
#Sta/Elev= 30
  3160.1 1660.75  3248.4 1659.16  3400.8 1652.56  3522.7 1648.72  3600.5 1647.78
  3659.4 1645.77  3868.1 1642.91  4812.8 1642.81  4894.1 1644.57  4914.9 1643.60
  4934.7 1640.07  4944.9 1641.91  4955.0 1639.69  4963.7 1636.75  4968.7 1637.27
  4975.3 1634.59  4977.2 1631.14  4977.7 1630.64  5009.1 1631.14  5013.7 1633.38
  5026.6 1634.09  5036.9 1637.57  5060.1 1642.42  5067.8 1642.96  5096.2 1640.58
  5170.9 1645.28  5243.0 1655.89  5335.8 1662.62  5356.4 1665.28  5408.0 1668.05
#Mann=3,-1,0
  3160.1    0.05       0  4977.2    0.07       0  5009.1    0.12       0
Bank Sta=4977.2,5009.1
Exp/Cntr=0.3,0.1

Type RM Length L Ch R = 1,58988,539,539,539
BEGIN DESCRIPTION:
Deadman Creek 66.0
END DESCRIPTION:
XS GIS Cut Line= 3
      1616707.76      6906594.45      1618605.00      6906738.00
      1619054.99      6906538.00
#Sta/Elev= 30
  3096.4 1652.48  3444.6 1649.48  3484.8 1647.55  3645.2 1644.53  3765.6 1644.76
  3936.0 1642.10  4139.6 1642.65  4226.9 1641.09  4357.2 1640.97  4407.5 1637.93
  4477.6 1640.16  4688.2 1642.32  4888.8 1641.96  4918.8 1642.99  4969.0 1638.53
  4989.0 1632.35  4998.7 1631.27  4999.2 1630.77  5030.7 1631.27  5031.2 1632.51
  5036.7 1631.27  5042.8 1635.44  5053.8 1638.66  5106.3 1642.35  5180.9 1642.97
  5226.0 1643.49  5332.2 1646.91  5355.4 1652.50  5371.1 1654.36  5491.5 1662.26
#Mann=6,-1,0
  3096.4    0.05       0  4998.7    0.05       0  5030.7    0.05       0
  5106.3    0.05       0  5180.9    0.12       0  5226.0    0.05       0
Bank Sta=4998.7,5030.7
Exp/Cntr=0.3,0.1

Type RM Length L Ch R = 1,58449,547,547,547
BEGIN DESCRIPTION:
Deadman Creek 65.0
END DESCRIPTION:
XS GIS Cut Line= 3
      1616423.03      6907115.28      1618455.00      6907238.00
      1619339.65      6906768.06
#Sta/Elev= 30
  2953.7 1658.15  3707.0 1643.61  3857.3 1643.63  3917.4 1642.04  4538.6 1641.35
  4638.7 1640.03  4698.8 1636.57  4819.1 1640.42  4959.3 1641.04  4992.2 1638.85
  4997.5 1635.13  5003.2 1636.24  5019.5 1632.72  5025.2 1635.01  5039.8 1635.23
  5047.2 1636.08  5053.1 1631.19  5053.6 1630.69  5085.1 1631.19  5091.3 1638.09
  5101.8 1640.17  5123.8 1641.75  5153.6 1641.69  5403.9 1640.81  5579.7 1643.16
  5601.7 1644.99  5634.3 1650.86  5771.9 1659.37  5876.1 1662.62  5991.1 1662.85
#Mann=5,-1,0
  2953.7    0.05       0  5039.8    0.12       0  5053.1    0.05       0
  5085.1    0.12       0  5153.6    0.05       0
Bank Sta=5053.1,5085.1
Exp/Cntr=0.3,0.1

Type RM Length L Ch R = 1,57902,566,566,566
BEGIN DESCRIPTION:
Deadman Creek 64.0
END DESCRIPTION:
XS GIS Cut Line= 3
      1616541.02      6908261.12      1618405.00      6907738.00
      1619205.02      6906937.98
#Sta/Elev= 30
  3058.4 1650.43  3104.1 1650.74  3613.0 1645.01  3997.3 1644.23  4329.7 1645.56
  4475.1 1645.13  4757.3 1641.03  4890.5 1640.02  4911.3 1638.69  4943.3 1639.85
  4963.2 1637.62  4974.4 1635.14  4977.4 1635.19  4985.5 1630.63  4986.0 1630.13
  5018.2 1630.63  5022.7 1632.13  5036.8 1631.20  5051.0 1638.38  5065.1 1639.41
  5110.6 1639.71  5390.4 1640.84  5644.9 1639.38  5871.2 1642.13  5913.6 1643.34
  5956.1 1650.12  5984.3 1652.91  6012.6 1654.81  6083.3 1656.56  6125.8 1659.41
#Mann=5,-1,0
  3058.4    0.05       0  4974.4    0.12       0  4985.5    0.07       0
  5018.2    0.12       0  5110.6    0.05       0
Bank Sta=4985.5,5018.2
Exp/Cntr=0.3,0.1

Type RM Length L Ch R = 1,57336,522,522,522
BEGIN DESCRIPTION:
Deadman Creek 63.0
END DESCRIPTION:
XS GIS Cut Line= 3
      1617751.05      6908731.97      1618755.00      6908138.00
      1620120.40      6907109.04
#Sta/Elev= 30
  3827.6 1644.33  4299.8 1644.76  4773.7 1640.13  4943.4 1639.97  4980.5 1639.16
  4991.2 1637.07  4997.2 1637.07  4999.6 1630.81  5000.1 1630.31  5032.3 1630.81
  5057.6 1631.03  5065.9 1633.20  5072.2 1637.57  5086.7 1640.19  5101.3 1640.08
  5107.6 1638.87  5186.7 1637.92  5394.8 1638.72  5494.8 1637.46  5850.8 1639.86
  6000.7 1642.23  6100.7 1644.65  6136.1 1646.46  6208.7 1647.37  6250.6 1648.67
  6321.4 1653.07  6379.6 1655.21  6515.0 1658.24  6558.7 1659.97  6703.8 1662.70
#Mann=3,-1,0
  3827.6    0.05       0  4999.6    0.05       0  5032.3    0.05       0
Bank Sta=4999.6,5032.3
Exp/Cntr=0.3,0.1

Type RM Length L Ch R = 1,56814,1801,1801,1801
BEGIN DESCRIPTION:
Deadman Creek 62.0
END DESCRIPTION:
XS GIS Cut Line= 3
      1617336.52      6909122.61      1619205.00      6908388.00
      1620304.96      6907538.03
#Sta/Elev= 30
  3003.9 1645.79  4070.1 1642.93  4356.2 1639.93  4571.1 1640.67  4743.0 1638.38
  4863.9 1638.60  4882.7 1637.91  4904.2 1634.90  4957.9 1633.90  4966.9 1631.96
  4971.8 1628.69  4972.4 1628.19  5001.4 1628.69  5002.1 1634.90  5008.9 1639.55
  5018.9 1640.27  5047.8 1638.38  5211.8 1636.35  5496.1 1637.58  5525.1 1638.63
  5753.3 1640.55  5788.6 1641.89  5832.1 1649.30  5867.4 1652.27  5952.6 1655.89
  5967.1 1657.68  5987.9 1657.60  6060.3 1661.08  6066.7 1660.28  6401.7 1668.21
#Mann=3,-1,0
  3003.9    0.05       0  4971.8    0.05       0  5001.4    0.05       0
Bank Sta=4971.8,5001.4
Exp/Cntr=0.3,0.1

Type RM Length L Ch R = 1,55013,1249,1249,1249
BEGIN DESCRIPTION:
Mapping XS 79f90c0c
END DESCRIPTION:
XS GIS Cut Line= 3
      1618150.25      6909096.31      1619732.31      6909244.52
      1620590.30      6908376.20
#Sta/Elev= 30
  2669.6 1643.15  3106.3 1641.69  3297.1 1641.53  3417.6 1642.50  3508.0 1640.78
  3548.2 1641.92  3789.2 1640.63  3960.0 1640.62  4350.0 1637.40  4555.0 1637.68
  4647.0 1638.73  4873.2 1634.85  4908.6 1635.55  4922.7 1634.90  4943.9 1632.13
  4976.8 1630.82  4977.4 1630.32  5009.4 1630.32  5010.0 1630.82  5035.9 1631.51
  5099.5 1636.14  5125.2 1636.14  5149.0 1636.82  5156.0 1637.88  5170.2 1640.57
  5177.3 1643.30  5198.5 1649.09  5205.6 1649.54  5304.6 1652.67  5479.3 1654.04
#Mann=4,-1,0
  2669.6    0.05       0  4976.8    0.07       0  5010.0    0.05       0
  5125.2    0.05       0
Bank Sta=4976.8,5010
Exp/Cntr=0.3,0.1

Type RM Length L Ch R = 1,53764,229,229,229
BEGIN DESCRIPTION:
Mapping XS 1688a6f5
END DESCRIPTION:
XS GIS Cut Line= 3
      1618155.97      6909143.42      1620551.83      6909365.65
      1621579.64      6909407.32
#Sta/Elev= 30
  1987.6 1643.16  2609.3 1641.59  2729.8 1642.78  2770.0 1641.17  2820.2 1641.99
  3322.3 1640.48  4035.3 1636.06  4573.6 1634.13  4717.2 1635.14  4867.3 1634.26
  4887.3 1634.00  4917.3 1632.18  4957.4 1627.36  4967.4 1624.13  4970.3 1624.08
  4971.0 1623.58  5004.5 1624.08  5027.4 1630.62  5037.4 1634.42  5047.4 1636.24
  5065.7 1638.69  5070.7 1638.24  5117.5 1640.87  5147.5 1644.78  5167.5 1649.00
  5197.6 1652.34  5267.6 1655.20  5307.7 1657.81  5397.7 1659.59  5422.4 1659.28
#Mann=3,-1,0
  1987.6    0.05       0  4970.3    0.05       0  5004.5    0.05       0
Bank Sta=4970.3,5004.5
Exp/Cntr=0.3,0.1

Type RM Length L Ch R = 1,53535,605,605,605
BEGIN DESCRIPTION:
Mapping XS c0c2f554
END DESCRIPTION:
XS GIS Cut Line= 2
      1619378.21      6909442.04      1621550.93      6909587.81
#Sta/Elev= 30
  3086.2 1641.65  3143.1 1641.22  3213.3 1642.03  3249.2 1640.65  3363.6 1640.57
  3399.0 1639.57  3423.7 1640.33  3548.9 1638.15  3594.1 1636.55  3624.2 1636.99
  3985.0 1635.29  4443.0 1634.61  4716.6 1633.04  4867.0 1632.72  4887.0 1633.60
  4917.1 1633.42  4937.1 1632.15  4995.2 1623.29  4995.9 1622.79  5029.4 1623.29
  5042.5 1631.18  5047.5 1628.44  5057.4 1632.29  5067.4 1634.96  5107.5 1641.51
  5116.6 1644.19  5147.6 1650.61  5157.6 1651.53  5217.8 1652.27  5263.8 1651.95
#Mann=4,-1,0
  3086.2    0.05       0  4995.2    0.03       0  5029.4    0.05       0
  5116.6    0.12       0
Bank Sta=4995.2,5029.4
Exp/Cntr=0.3,0.1

Type RM Length L Ch R = 1,52930,547,547,547
BEGIN DESCRIPTION:
Deadman Creek 56.0
END DESCRIPTION:
XS GIS Cut Line= 3
      1619371.30      6910067.04      1621455.00      6910088.00
      1622055.02      6909988.00
#Sta/Elev= 30
  2915.6 1639.83  3069.3 1639.93  3129.3 1638.70  3339.3 1638.86  3359.3 1637.17
  3389.3 1637.94  3489.3 1636.59  3519.3 1634.89  3669.3 1633.72  4479.4 1633.75
  4679.4 1630.41  4939.4 1634.20  4979.4 1633.53  4989.4 1629.12  4996.9 1623.15
  5001.9 1623.15  5002.3 1621.47  5003.0 1620.97  5033.1 1621.47  5040.0 1625.08
  5088.1 1626.03  5100.8 1625.37  5121.1 1627.56  5141.3 1631.69  5162.7 1633.80
  5176.1 1633.58  5222.4 1633.52  5270.6 1637.38  5374.5 1642.55  5607.7 1649.17
#Mann=5,-1,0
  2915.6    0.05       0  5002.3    0.03       0  5033.1    0.05       0
  5162.7    0.12       0  5176.1    0.05       0
Bank Sta=5002.3,5033.1
Exp/Cntr=0.3,0.1

Type RM Length L Ch R = 1,52383,584,584,584
BEGIN DESCRIPTION:
Deadman Creek 55.0
END DESCRIPTION:
XS GIS Cut Line= 4
      1619987.55      6911169.43      1621571.99      6910625.15
      1621705.00      6910538.00      1622104.97      6910388.01
#Sta/Elev= 30
  3166.1 1640.44  3338.8 1634.34  3432.6 1633.49  3533.5 1630.76  3544.1 1630.75
  3557.6 1632.89  3588.8 1629.38  3620.1 1630.31  3828.3 1629.88  3927.3 1631.15
  4273.6 1632.01  4510.5 1629.44  4661.5 1632.15  4914.5 1633.32  4935.6 1631.55
  4950.7 1626.62  4959.1 1619.80  4959.7 1619.30  4990.2 1619.80  4992.9 1626.14
  4997.4 1626.68  5032.5 1623.39  5053.8 1625.44  5070.7 1624.35  5095.7 1625.38
  5107.2 1627.48  5150.0 1631.85  5161.5 1634.83  5190.9 1637.08  5427.6 1652.22
#Mann=4,-1,0
  3166.1    0.05       0  4959.1    0.07       0  4990.2    0.05       0
  5190.9    0.05       0
Bank Sta=4959.1,4990.2
Exp/Cntr=0.3,0.1

Type RM Length L Ch R = 1,51799,537,537,537
BEGIN DESCRIPTION:
Deadman Creek 54.0
END DESCRIPTION:
XS GIS Cut Line= 3
      1620455.05      6911487.99      1622055.00      6910988.00
      1622405.03      6910787.98
#Sta/Elev= 30
  3323.3 1644.71  3372.0 1636.43  3377.2 1636.47  3404.4 1632.22  3436.9 1631.08
  3449.0 1628.62  3480.4 1631.95  3507.1 1628.66  3512.4 1629.61  3539.6 1628.81
  3857.6 1628.42  4242.6 1631.52  4894.8 1632.10  4936.7 1630.95  4945.6 1629.00
  4950.8 1626.57  4957.6 1618.32  4966.6 1618.29  4967.3 1617.79  5004.6 1618.29
  5007.5 1623.79  5013.2 1626.21  5034.8 1631.02  5066.5 1630.21  5131.3 1631.49
  5160.8 1635.29  5255.1 1644.48  5308.4 1647.99  5351.6 1652.17  5402.7 1654.53
#Mann=3,-1,0
  3323.3    0.05       0  4966.6    0.07       0  5004.6    0.12       0
Bank Sta=4966.6,5004.6
Exp/Cntr=0.3,0.1

Type RM Length L Ch R = 1,51262,546,546,546
BEGIN DESCRIPTION:
Deadman Creek 53.0
END DESCRIPTION:
XS GIS Cut Line= 3
      1620204.96      6911588.00      1622405.00      6911388.00
      1622604.99      6911038.03
#Sta/Elev= 30
  2796.0 1657.19  2846.3 1657.17  2936.6 1654.42  3037.0 1648.20  3087.2 1643.20
  3117.4 1637.76  3157.5 1632.73  3187.7 1630.98  3207.7 1628.42  3217.8 1628.25
  3247.9 1631.45  3257.9 1629.52  3278.0 1628.04  3770.0 1630.46  4894.7 1630.80
  4924.8 1630.50  4934.8 1629.04  4954.9 1618.85  4967.7 1617.33  4968.4 1616.83
  5002.3 1617.33  5002.6 1623.17  5028.2 1624.45  5040.4 1628.53  5072.1 1630.26
  5077.8 1633.75  5099.4 1637.77  5132.9 1639.40  5298.1 1651.80  5408.2 1656.45
#Mann=4,-1,0
  2796.0    0.05       0  4967.7    0.07       0  5002.3    0.05       0
  5132.9    0.05       0
Bank Sta=4967.7,5002.3
Exp/Cntr=0.3,0.1

Type RM Length L Ch R = 1,50716,565,565,565
BEGIN DESCRIPTION:
Deadman Creek 52.0
END DESCRIPTION:
XS GIS Cut Line= 3
      1620354.98      6911688.00      1622555.00      6911888.00
      1622905.00      6912088.00
#Sta/Elev= 30
  2791.0 1655.87  2971.8 1644.05  3042.0 1632.04  3132.4 1627.53  3152.5 1630.38
  3182.6 1627.11  3433.7 1629.78  4086.3 1629.26  4618.5 1630.16  4678.8 1631.65
  4789.2 1628.01  4908.8 1629.43  4929.8 1629.32  4939.8 1620.74  4949.9 1622.13
  4970.0 1619.11  4972.7 1616.76  4973.4 1616.26  5007.4 1616.76  5008.0 1619.29
  5013.8 1617.50  5029.6 1622.16  5051.2 1624.78  5067.0 1633.44  5072.8 1633.36
  5080.7 1636.99  5094.2 1637.15  5110.2 1641.04  5218.9 1651.29  5403.2 1661.29
#Mann=5,-1,0
  2791.0    0.05       0  4908.8    0.12       0  4972.7    0.07       0
  5007.4    0.12       0  5094.2    0.05       0
Bank Sta=4972.7,5007.4
Exp/Cntr=0.3,0.1

Type RM Length L Ch R = 1,50151,734,734,734
BEGIN DESCRIPTION:
Deadman Creek 51.0
END DESCRIPTION:
XS GIS Cut Line= 3
      1620316.24      6912424.31      1622505.00      6912438.00
      1622904.99      6912388.00
#Sta/Elev= 30
  2811.2 1651.02  2980.0 1649.79  3130.0 1644.30  3210.0 1630.05  3320.0 1625.69
  3410.0 1628.39  3480.0 1624.64  3550.0 1627.37  4860.0 1627.39  4890.0 1632.09
  4900.0 1631.98  4920.0 1627.61  4940.0 1627.27  4961.5 1623.37  4970.0 1618.19
  4982.6 1616.42  4983.3 1615.92  5017.4 1616.42  5020.2 1616.42  5030.2 1621.92
  5050.4 1624.57  5060.5 1627.56  5080.6 1636.44  5107.8 1641.27  5118.4 1644.25
  5123.5 1643.94  5151.2 1648.68  5231.8 1654.90  5302.3 1658.61  5403.1 1661.07
#Mann=5,-1,0
  2811.2    0.05       0  4961.5    0.12       0  4982.6    0.07       0
  5017.4    0.12       0  5107.8    0.05       0
Bank Sta=4982.6,5017.4
Exp/Cntr=0.3,0.1

Type RM Length L Ch R = 1,49417,1217,1217,1217
BEGIN DESCRIPTION:
Mapping XS 75bef355
END DESCRIPTION:
XS GIS Cut Line= 4
      1620607.86      6913221.18      1622165.19      6913122.22
      1622399.56      6913101.39      1622784.69      6912882.80
#Sta/Elev= 30
  3299.1 1650.07  3742.8 1636.66  3807.3 1630.78  3837.3 1626.28  3887.4 1623.50
  3957.6 1623.24  4007.7 1625.03  4027.7 1627.24  4047.7 1623.11  4060.8 1623.20
  4067.8 1624.43  4087.8 1625.25  4879.5 1625.71  4919.6 1627.03  4964.3 1626.35
  4969.8 1622.06  4979.9 1616.61  4990.7 1616.15  4991.0 1616.15  4991.8 1615.65
  5032.8 1616.15  5050.1 1621.30  5070.2 1624.28  5205.3 1628.50  5238.5 1631.04
  5276.6 1636.19  5301.7 1637.72  5438.2 1645.41  5534.8 1648.56  5537.7 1649.39
#Mann=7,-1,0
  3299.1    0.05       0  4990.7    0.12       0  4991.0    0.07       0
  5032.8    0.12       0  5205.3    0.05       0  5238.5    0.12       0
  5301.7    0.05       0
Bank Sta=4991,5032.8
Exp/Cntr=0.3,0.1

Type RM Length L Ch R = 1,48200,769,769,769
BEGIN DESCRIPTION:
Deadman Creek 50.0
END DESCRIPTION:
XS GIS Cut Line= 3
      1621201.62      6914242.03      1621706.85      6913887.85
      1623279.77      6913080.56
#Sta/Elev= 30
  4380.1 1638.27  4536.0 1633.39  4571.8 1630.28  4601.4 1623.93  4622.3 1624.62
  4637.1 1619.27  4679.0 1621.09  4693.8 1620.10  4708.6 1615.63  4714.7 1617.92
  4723.4 1615.99  4729.6 1619.45  4744.4 1619.90  4794.9 1617.19  4815.8 1622.41
  4860.3 1624.31  4887.3 1623.46  4923.1 1618.75  4973.6 1621.46  5004.2 1617.49
  5008.1 1614.60  5008.7 1614.10  5039.4 1614.60  5062.5 1620.44  5120.8 1620.80
  5181.7 1625.44  5902.7 1625.76  6318.7 1630.90  6429.7 1638.75  6765.1 1648.20
#Mann=3,-1,0
  4380.1    0.05       0  5008.1    0.05       0  5039.4    0.05       0
Bank Sta=5008.1,5039.4
Exp/Cntr=0.3,0.1

Type RM Length L Ch R = 1,47431,570,570,570
BEGIN DESCRIPTION:
Deadman Creek 49.0
END DESCRIPTION:
XS GIS Cut Line= 3
      1621805.00      6914937.96      1621855.00      6914538.00
      1623405.02      6913087.98
#Sta/Elev= 30
  4596.8 1656.47  4720.2 1650.28  4788.2 1645.54  4818.5 1642.00  4848.7 1640.30
  4889.0 1634.61  4929.3 1632.02  4962.1 1620.83  4989.8 1615.31  4992.2 1612.83
  4992.8 1612.33  5017.6 1612.83  5021.1 1615.36  5042.1 1615.46  5063.6 1619.38
  5134.4 1624.04  5240.5 1621.97  5396.3 1621.38  5594.1 1623.47  6174.5 1624.30
  6584.8 1627.46  6634.1 1630.49  6669.8 1636.43  6719.1 1640.75  6839.3 1644.53
  6952.6 1646.88  6973.6 1646.05  6981.0 1647.53  7051.8 1651.99  7122.4 1654.56
#Mann=3,-1,0
  4596.8    0.05       0  4992.2    0.05       0  5017.6    0.05       0
Bank Sta=4992.2,5017.6
Exp/Cntr=0.3,0.1

Type RM Length L Ch R = 1,46861,597,597,597
BEGIN DESCRIPTION:
Deadman Creek 48.0
END DESCRIPTION:
XS GIS Cut Line= 3
      1622355.00      6915138.03      1622355.00      6914738.00
      1623455.01      6913137.99
#Sta/Elev= 30
  4599.7 1655.48  4709.7 1650.08  4739.7 1646.88  4909.7 1635.15  4919.7 1633.88
  4939.7 1625.28  4959.7 1619.03  4974.4 1611.69  4975.3 1611.19  5007.1 1611.69
  5007.2 1614.88  5013.2 1614.76  5022.1 1616.62  5114.7 1619.06  5129.6 1620.93
  5294.0 1619.20  5359.7 1621.44  5524.0 1623.05  5783.8 1623.23  5804.8 1624.20
  5825.8 1623.19  6019.9 1623.68  6395.3 1626.58  6473.9 1629.86  6524.6 1636.03
  6560.5 1638.87  6668.1 1642.43  6689.0 1644.24  6820.0 1646.68  6941.4 1653.72
#Mann=3,-1,0
  4599.7    0.05       0  4974.4    0.05       0  5007.1    0.05       0
Bank Sta=4974.4,5007.1
Exp/Cntr=0.3,0.1

Type RM Length L Ch R = 1,46264,659,659,659
BEGIN DESCRIPTION:
Deadman Creek 47.0
END DESCRIPTION:
XS GIS Cut Line= 3
      1622654.98      6915038.02      1622904.77      6914689.93
      1623654.98      6913088.04
#Sta/Elev= 30
  4570.0 1649.12  4663.4 1643.78  4841.4 1637.07  4850.0 1634.30  4870.9 1632.19
  4885.6 1625.47  4891.8 1626.51  4900.3 1624.19  4906.5 1624.65  4921.2 1618.25
  4927.4 1618.97  4936.0 1615.64  4942.1 1616.11  4950.7 1611.30  4956.8 1612.83
  4959.0 1611.09  4960.0 1610.59  5014.0 1611.09  5022.7 1616.78  5031.3 1619.05
  5054.1 1619.89  6074.5 1624.94  6104.8 1627.64  6114.6 1626.45  6171.3 1634.94
  6239.8 1640.03  6547.7 1643.94  6633.5 1648.69  6684.7 1653.58  6767.3 1658.77
#Mann=3,-1,0
  4570.0    0.05       0  4959.0    0.05       0  5014.0    0.05       0
Bank Sta=4959,5014
Exp/Cntr=0.3,0.1

Type RM Length L Ch R = 1,45605,517,517,517
BEGIN DESCRIPTION:
Deadman Creek 46.0
END DESCRIPTION:
XS GIS Cut Line= 3
      1622905.01      6915037.99      1623472.48      6914518.06
      1624104.99      6913738.02
#Sta/Elev= 30
  4222.3 1642.38  4300.3 1638.52  4321.3 1635.65  4378.0 1631.35  4420.5 1624.41
  4455.7 1621.78  4540.8 1619.64  4561.7 1620.92  4604.3 1619.65  4668.4 1620.79
  4675.2 1618.40  4682.6 1619.56  4689.4 1616.72  4703.6 1616.24  4859.6 1616.66
  4908.9 1614.45  4951.5 1615.48  4958.2 1613.77  4979.8 1613.02  4985.6 1609.07
  4986.3 1608.57  5014.8 1609.07  5029.9 1619.22  5079.5 1620.96  5547.9 1621.72
  5704.5 1623.75  5739.7 1626.90  5803.7 1640.47  5826.0 1643.11  5996.2 1656.10
#Mann=3,-1,0
  4222.3    0.05       0  4985.6    0.03       0  5014.8    0.05       0
Bank Sta=4985.6,5014.8
Exp/Cntr=0.3,0.1

Type RM Length L Ch R = 1,45088,489,489,489
BEGIN DESCRIPTION:
Deadman Creek 45.0
END DESCRIPTION:
XS GIS Cut Line= 3
      1623005.00      6915138.00      1623909.98      6914835.77
      1624628.71      6914143.08
#Sta/Elev= 30
  4314.1 1641.63  4361.5 1639.16  4366.8 1637.83  4393.1 1636.10  4503.9 1621.74
  4525.0 1622.98  4535.5 1621.24  4556.6 1620.60  4835.5 1618.51  4925.0 1614.97
  4946.7 1616.12  4956.6 1613.78  4961.9 1614.24  4967.8 1609.27  4968.1 1607.61
  4968.8 1607.11  4997.3 1607.61  4999.4 1610.64  5031.0 1611.15  5051.4 1613.12
  5119.9 1614.24  5125.9 1615.86  5177.8 1620.56  5454.2 1620.01  5991.6 1622.67
  6026.8 1625.70  6097.6 1640.34  6140.0 1644.77  6210.8 1649.35  6266.4 1651.14
#Mann=3,-1,0
  4314.1    0.05       0  4968.1    0.03       0  4997.3    0.05       0
Bank Sta=4968.1,4997.3
Exp/Cntr=0.3,0.1

Type RM Length L Ch R = 1,44599,365,365,365
BEGIN DESCRIPTION:
Deadman Creek 44.0
END DESCRIPTION:
XS GIS Cut Line= 3
      1623405.03      6915587.98      1623805.00      6915338.00
      1625204.97      6915238.00
#Sta/Elev= 30
  4527.9 1640.63  4556.8 1637.29  4593.3 1628.99  4614.5 1626.60  4629.9 1622.06
  4693.5 1619.51  4955.3 1615.15  4976.6 1614.05  4991.9 1611.22  4997.1 1606.35
  4997.8 1605.85  5026.3 1606.35  5029.6 1611.88  5039.7 1615.51  5059.7 1616.86
  5067.2 1619.33  5212.6 1619.87  5370.5 1617.16  5480.8 1618.37  5540.9 1614.92
  5791.6 1618.96  5952.0 1618.92  6122.4 1621.10  6172.5 1624.21  6190.1 1628.61
  6195.1 1628.30  6232.7 1638.73  6272.8 1645.97  6343.0 1652.65  6403.1 1655.65
#Mann=3,-1,0
  4527.9    0.05       0  4997.1    0.05       0  5026.3    0.05       0
Bank Sta=4997.1,5026.3
Exp/Cntr=0.3,0.1

Type RM Length L Ch R = 1,44234,1063,1063,1063
BEGIN DESCRIPTION:
Deadman Creek 43.0
END DESCRIPTION:
XS GIS Cut Line= 3
      1623191.23      6915799.31      1623816.23      6915700.35
      1625481.43      6915460.98
#Sta/Elev= 30
  4365.5 1650.33  4622.4 1642.97  4652.8 1639.62  4733.8 1621.39  4981.6 1617.32
  4994.0 1605.42  4994.9 1604.92  5030.6 1605.42  5048.5 1611.82  5067.8 1613.35
  5088.0 1608.89  5108.2 1615.76  5148.6 1617.94  5178.9 1617.18  5199.1 1611.66
  5219.3 1610.43  5249.6 1613.58  5291.1 1613.02  5310.2 1611.92  5328.2 1614.27
  5522.4 1618.73  6118.4 1621.47  6199.3 1640.23  6310.2 1652.30  6411.4 1656.13
  6456.2 1660.68  6492.3 1656.52  6532.7 1655.63  6603.4 1662.34  6680.6 1664.54
#Mann=5,-1,0
  4365.5    0.05       0  4994.0    0.05       0  5030.6    0.05       0
  5048.5    0.12       0  5291.1    0.05       0
Bank Sta=4994,5030.6
Exp/Cntr=0.3,0.1

Type RM Length L Ch R = 1,43171,654,654,654
BEGIN DESCRIPTION:
Deadman Creek 42.0
END DESCRIPTION:
XS GIS Cut Line= 3
      1623205.04      6916538.00      1624165.19      6916590.97
      1624847.48      6917090.98
#Sta/Elev= 30
  4499.4 1664.20  4609.5 1659.69  4639.6 1657.61  4669.6 1656.98  4699.7 1653.63
  4749.7 1651.11  4768.2 1648.57  4839.9 1643.40  4849.9 1641.79  4869.9 1635.10
  4910.0 1625.13  4920.0 1620.94  4940.0 1610.27  4949.1 1608.09  4980.1 1603.77
  4983.7 1601.38  4984.4 1600.38  5015.7 1600.38  5016.5 1601.38  5020.2 1614.05
  5060.2 1612.56  5110.3 1613.77  5135.0 1612.28  5210.4 1615.23  5310.6 1617.07
  5795.5 1619.28  5988.3 1621.40  6109.5 1623.88  6253.8 1628.41  6306.9 1628.63
#Mann=3,-1,0
  4499.4    0.05       0  4983.7    0.05       0  5016.5    0.05       0
Bank Sta=4983.7,5016.5
Exp/Cntr=0.3,0.1

Type RM Length L Ch R = 1,42517,655,655,655
BEGIN DESCRIPTION:
Deadman Creek 41.0
END DESCRIPTION:
XS GIS Cut Line= 3
      1623378.76      6917158.68      1623705.00      6917188.00
      1624915.17      6917325.35
#Sta/Elev= 30
  4672.0 1648.94  4798.8 1644.97  4832.9 1642.32  4859.0 1637.83  4889.1 1629.61
  4909.2 1624.94  4929.3 1615.03  4939.0 1613.08  4944.0 1613.31  4969.4 1606.63
  4980.3 1600.59  4981.4 1599.59  5025.2 1599.59  5026.3 1600.59  5029.7 1606.72
  5039.3 1612.37  5040.6 1612.42  5049.9 1613.86  5059.9 1614.27  5100.2 1612.72
  5432.3 1617.25  5653.7 1618.63  5865.1 1623.51  6015.2 1627.78  6046.2 1628.04
  6076.4 1629.36  6109.8 1629.27  6156.9 1629.95  6187.1 1631.13  6217.5 1631.01
#Mann=4,-1,0
  4672.0    0.05       0  4980.3    0.07       0  5026.3    0.05       0
  5040.6    0.05       0
Bank Sta=4980.3,5026.3
Exp/Cntr=0.3,0.1

Type RM Length L Ch R = 1,41862,679,679,679
BEGIN DESCRIPTION:
Deadman Creek 40.0
END DESCRIPTION:
XS GIS Cut Line= 3
      1623237.62      6917573.99      1623866.07      6917789.26
      1624741.65      6917840.88
#Sta/Elev= 30
  4346.7 1635.04  4386.2 1633.83  4460.2 1629.01  4502.9 1624.51  4523.6 1623.50
  4534.2 1620.91  4565.9 1618.28  4773.8 1611.82  4798.5 1612.14  4830.2 1610.03
  4902.9 1609.62  4930.3 1610.19  4946.4 1608.06  4967.6 1606.78  4978.2 1605.19
  4987.5 1598.61  4988.3 1597.61  5019.6 1597.61  5020.3 1598.61  5030.0 1612.77
  5040.0 1615.38  5050.0 1615.97  5106.2 1613.03  5120.1 1612.50  5320.5 1617.01
  5611.0 1621.16  5755.2 1624.47  5851.4 1628.60  5871.4 1627.65  5888.1 1628.41
#Mann=5,-1,0
  4346.7    0.05       0  4902.9    0.12       0  4987.5    0.07       0
  5020.3    0.12       0  5106.2    0.05       0
Bank Sta=4987.5,5020.3
Exp/Cntr=0.3,0.1

Type RM Length L Ch R = 1,41183,777,777,777
BEGIN DESCRIPTION:
Deadman Creek 39.0
END DESCRIPTION:
XS GIS Cut Line= 4
      1623004.98      6917587.96      1623216.76      6918136.48
      1623909.98      6918419.10      1624471.20      6918621.76
#Sta/Elev= 30
  3668.0 1637.09  3786.0 1631.25  3861.0 1622.59  3955.8 1617.58  4515.2 1611.50
  4860.1 1613.15  4878.8 1608.12  4884.2 1609.73  4891.2 1604.33  4902.0 1600.52
  4932.3 1603.08  4937.7 1600.97  4956.0 1603.73  4974.2 1597.79  4974.9 1596.79
  5007.0 1597.79  5007.8 1599.35  5009.9 1603.45  5015.7 1606.67  5046.3 1608.16
  5063.1 1611.57  5194.4 1611.33  5319.1 1615.40  5360.8 1616.17  5382.1 1611.93
  5392.7 1617.47  5423.8 1625.28  5435.2 1630.50  5485.1 1639.21  5601.3 1650.65
#Mann=5,-1,0
  3668.0    0.05       0  4974.2    0.03       0  5007.0    0.05       0
  5007.8    0.12       0  5319.1    0.05       0
Bank Sta=4974.2,5007
Exp/Cntr=0.3,0.1

Type RM Length L Ch R = 1,40406,695,695,695
BEGIN DESCRIPTION:
Deadman Creek 38.0
END DESCRIPTION:
XS GIS Cut Line= 3
      1621954.99      6917688.00      1623755.00      6919088.00
      1624154.97      6919487.97
#Sta/Elev= 30
  2725.5 1654.98  2925.5 1649.39  3118.2 1639.88  3244.9 1635.51  3367.1 1626.96
  3387.9 1624.10  3630.4 1616.98  4136.2 1610.81  4171.5 1611.83  4229.5 1610.20
  4478.3 1612.78  4899.1 1612.26  4913.6 1611.76  4928.0 1609.27  4955.2 1602.06
  4963.3 1601.85  4969.7 1594.84  4970.9 1594.84  4971.7 1593.84  5003.0 1593.84
  5003.8 1594.84  5005.9 1602.45  5009.4 1602.45  5034.1 1619.37  5048.3 1625.98
  5090.7 1640.25  5104.9 1643.66  5147.3 1645.96  5458.4 1655.21  5571.5 1657.23
#Mann=3,-1,0
  2725.5    0.05       0  4970.9    0.05       0  5003.8    0.05       0
Bank Sta=4970.9,5003.8
Exp/Cntr=0.3,0.1

Type RM Length L Ch R = 1,39711,763,763,763
BEGIN DESCRIPTION:
Deadman Creek 37.0
END DESCRIPTION:
XS GIS Cut Line= 3
      1621955.02      6917788.02      1623155.00      6919388.00
      1623655.01      6919588.00
#Sta/Elev= 30
  3000.1 1653.57  3136.5 1649.61  3171.9 1647.07  3328.2 1640.70  3350.1 1638.53
  3450.1 1634.74  3571.9 1622.35  3657.4 1619.09  3863.6 1615.01  4386.5 1610.11
  4457.4 1608.23  4557.4 1611.35  4909.7 1610.92  4929.3 1610.52  4942.8 1610.02
  4957.7 1594.76  4958.7 1593.76  5002.6 1593.76  5003.6 1594.76  5009.5 1599.00
  5032.4 1600.61  5039.1 1601.65  5044.5 1604.06  5063.3 1606.97  5068.7 1612.63
  5098.4 1623.56  5183.2 1634.37  5278.8 1638.19  5301.6 1640.55  5538.6 1646.47
#Mann=5,-1,0
  3000.1    0.05       0  4909.7    0.12       0  4929.3    0.05       0
  4957.7    0.05       0  5003.6    0.05       0
Bank Sta=4957.7,5003.6
Exp/Cntr=0.3,0.1

Type RM Length L Ch R = 1,38948,862,862,862
BEGIN DESCRIPTION:
Mapping XS 338d8178
END DESCRIPTION:
XS GIS Cut Line= 4
      1621826.63      6918429.48      1622139.14      6919179.52
      1622701.64      6919986.81      1623341.11      6919695.67
#Sta/Elev= 30
  3557.0 1632.19  3652.9 1630.34  3698.7 1627.85  3804.9 1615.71  3858.7 1613.61
  4035.6 1611.75  4458.8 1610.56  4667.4 1607.18  4745.5 1609.53  4865.2 1609.06
  4896.8 1607.67  4911.7 1604.21  4917.8 1605.07  4940.5 1600.41  4977.1 1598.25
  4979.1 1594.68  4980.0 1593.68  5017.6 1593.68  5018.5 1594.68  5019.0 1596.48
  5025.8 1604.18  5033.8 1607.70  5062.4 1609.95  5108.4 1609.33  5313.9 1608.77
  5423.1 1606.94  5829.6 1611.30  5891.8 1614.53  5983.5 1627.08  6056.1 1634.55
#Mann=5,-1,0
  3557.0    0.05       0  4865.2    0.12       0  4979.1    0.07       0
  5018.5    0.12       0  5108.4    0.05       0
Bank Sta=4979.1,5018.5
Exp/Cntr=0.3,0.1

Type RM Length L Ch R = 1,38086,476,476,476
BEGIN DESCRIPTION:
Mapping XS 6e2b7662
END DESCRIPTION:
XS GIS Cut Line= 3
      1621363.08      6919986.80      1622378.73      6920200.35
      1623368.29      6919715.98
#Sta/Elev= 30
  4583.0 1635.85  4799.6 1631.87  4881.3 1625.98  4900.7 1622.13  4905.8 1622.73
  4942.6 1612.97  4950.5 1607.64  4955.6 1608.92  4973.3 1597.78  4976.4 1594.53
  4977.6 1593.53  5028.0 1593.53  5029.2 1594.53  5034.6 1600.01  5050.2 1606.17
  5077.6 1606.58  5235.1 1607.81  5388.9 1609.98  5588.3 1606.06  5716.9 1608.67
  5888.6 1609.01  6046.2 1606.86  6479.4 1610.86  6546.9 1613.29  6552.5 1614.94
  6585.3 1618.79  6607.6 1623.68  6636.9 1627.45  6681.9 1632.92  6722.6 1635.69
#Mann=5,-1,0
  4583.0    0.05       0  4976.4    0.05       0  5029.2    0.05       0
  5077.6    0.12       0  5235.1    0.05       0
Bank Sta=4976.4,5029.2
Exp/Cntr=0.3,0.1

Type RM Length L Ch R = 1,37610,705,705,705
BEGIN DESCRIPTION:
Deadman Creek 36.0
END DESCRIPTION:
XS GIS Cut Line= 3
      1621455.02      6920488.00      1621955.00      6920488.00
      1623554.97      6919688.02
#Sta/Elev= 30
  4505.6 1640.44  4805.6 1633.04  4855.6 1629.47  4865.6 1628.42  4875.6 1624.69
  4915.6 1614.39  4925.6 1610.58  4955.1 1594.41  4956.4 1593.41  5013.1 1593.41
  5014.5 1594.41  5019.6 1602.31  5036.3 1605.64  5050.1 1606.47  5076.5 1605.97
  5220.8 1607.65  5304.7 1605.77  5452.8 1605.85  5729.5 1610.05  5891.6 1607.00
  5936.3 1607.13  6400.3 1610.78  6428.3 1612.88  6445.1 1612.32  6467.4 1613.87
  6526.1 1626.34  6579.2 1633.35  6646.3 1640.04  6713.4 1645.11  6794.4 1647.28
#Mann=5,-1,0
  4505.6    0.05       0  4955.1    0.05       0  5014.5    0.05       0
  5050.1    0.12       0  5076.5    0.05       0
Bank Sta=4955.1,5014.5
Exp/Cntr=0.3,0.1

Type RM Length L Ch R = 1,36905,713,713,713
BEGIN DESCRIPTION:
Deadman Creek 35.0
END DESCRIPTION:
XS GIS Cut Line= 3
      1622105.00      6921387.99      1622405.00      6920988.00
      1623804.96      6920188.02
#Sta/Elev= 30
  4493.3 1639.69  4595.4 1637.31  4656.0 1635.91  4821.4 1627.71  4943.3 1617.29
  4986.0 1607.13  4990.2 1599.92  4996.2 1599.92  4996.9 1594.17  4998.6 1593.17
  5069.6 1594.17  5079.7 1595.34  5081.8 1596.51  5087.6 1603.65  5103.4 1605.05
  5187.8 1604.20  5522.4 1607.15  5638.3 1603.77  5711.0 1605.41  5776.5 1603.45
  5947.1 1607.04  6371.8 1609.73  6386.9 1611.01  6415.0 1618.85  6458.2 1633.06
  6474.0 1639.67  6489.8 1643.08  6502.1 1644.89  6533.0 1644.18  6605.7 1646.90
#Mann=6,-1,0
  4493.3    0.05       0  4595.4    0.12       0  4656.0    0.05       0
  4996.9    0.05       0  5069.6    0.05       0  5187.8    0.05       0
Bank Sta=4996.9,5069.6
Exp/Cntr=0.3,0.1

Type RM Length L Ch R = 1,36192,671,671,671
BEGIN DESCRIPTION:
Deadman Creek 34.0
END DESCRIPTION:
XS GIS Cut Line= 3
      1622354.98      6921588.01      1622955.00      6921388.00
      1623954.99      6920888.00
#Sta/Elev= 30
  4372.5 1635.87  4425.2 1630.63  4499.0 1626.20  4583.3 1613.72  4773.1 1603.47
  4783.6 1602.15  4795.5 1602.39  4825.8 1603.69  4920.6 1604.35  4941.7 1601.26
  4950.3 1593.80  4951.8 1592.80  5014.9 1592.80  5016.4 1593.80  5019.0 1594.89
  5027.3 1603.10  5059.0 1602.92  5130.8 1604.42  5287.3 1603.95  5429.8 1600.91
  5488.5 1602.65  5944.1 1605.52  6002.8 1607.77  6025.2 1613.00  6040.2 1618.20
  6047.5 1618.96  6055.9 1622.95  6092.3 1632.37  6109.0 1637.97  6123.0 1638.35
#Mann=6,-1,0
  4372.5    0.05       0  4795.5    0.12       0  4950.3    0.07       0
  5016.4    0.12       0  5059.0    0.05       0  6040.2    0.12       0
Bank Sta=4950.3,5016.4
Exp/Cntr=0.3,0.1

Type RM Length L Ch R = 1,35521,717,717,717
BEGIN DESCRIPTION:
Deadman Creek 33.0
END DESCRIPTION:
XS GIS Cut Line= 3
      1622702.83      6922261.50      1623205.00      6921988.00
      1624105.02      6921187.99
#Sta/Elev= 30
  4421.9 1635.44  4434.9 1635.55  4447.1 1633.00  4469.9 1630.97  4565.9 1624.91
  4582.1 1621.24  4617.9 1610.04  4647.6 1606.28  4816.6 1602.09  4942.0 1602.46
  4948.2 1601.22  4957.8 1593.40  4959.3 1592.40  5022.4 1592.40  5023.9 1593.40
  5035.9 1602.71  5071.9 1604.05  5397.2 1602.27  5482.5 1599.14  5582.0 1600.73
  5617.1 1602.95  5794.4 1601.73  5970.8 1604.14  5999.3 1606.22  6013.5 1608.95
  6070.4 1623.67  6084.6 1628.49  6113.0 1635.15  6141.4 1639.12  6197.9 1641.36
#Mann=3,-1,0
  4421.9    0.05       0  4957.8    0.03       0  5023.9    0.05       0
Bank Sta=4957.8,5023.9
Exp/Cntr=0.3,0.1

Type RM Length L Ch R = 1,34804,682,682,682
BEGIN DESCRIPTION:
Deadman Creek 32.0
END DESCRIPTION:
XS GIS Cut Line= 3
      1623191.22      6922820.15      1623405.00      6922638.00
      1624566.23      6921606.60
#Sta/Elev= 30
  4718.9 1629.47  4793.9 1629.07  4886.1 1621.51  4928.9 1612.19  4964.1 1595.42
  4973.8 1592.32  4975.3 1591.32  5038.4 1591.32  5039.9 1592.32  5042.0 1598.12
  5049.5 1599.12  5169.9 1600.07  5212.6 1602.47  5644.1 1600.04  5764.5 1600.71
  5800.5 1602.38  5899.2 1602.23  5970.2 1599.38  6012.9 1595.84  6033.8 1597.15
  6083.1 1596.65  6182.6 1602.39  6211.1 1609.20  6232.0 1610.59  6239.5 1612.52
  6274.6 1613.88  6317.3 1619.10  6366.6 1620.67  6466.1 1630.16  6552.9 1632.84
#Mann=3,-1,0
  4718.9    0.05       0  4973.8    0.05       0  5039.9    0.05       0
Bank Sta=4973.8,5039.9
Exp/Cntr=0.3,0.1

Type RM Length L Ch R = 1,34122,684,684,684
BEGIN DESCRIPTION:
Deadman Creek 31.0
END DESCRIPTION:
XS GIS Cut Line= 3
      1623705.02      6923587.95      1623905.00      6923088.00
      1624905.01      6922087.99
#Sta/Elev= 30
  4462.1 1636.04  4638.4 1628.10  4709.8 1621.81  4794.6 1608.92  4829.6 1595.17
  4871.3 1593.12  4892.9 1594.95  4925.2 1593.13  4979.0 1594.86  4985.8 1593.98
  4986.9 1591.05  4987.8 1590.05  5025.6 1590.05  5026.5 1591.05  5028.9 1594.04
  5057.1 1599.91  5071.3 1600.32  5255.1 1597.75  5340.0 1599.01  5424.8 1597.80
  5566.3 1600.18  5863.2 1600.85  5948.1 1599.78  5990.5 1594.60  6032.9 1597.41
  6188.5 1599.44  6230.9 1602.44  6287.5 1615.81  6344.1 1622.15  6414.8 1627.41
#Mann=3,-1,0
  4462.1    0.05       0  4986.9    0.05       0  5026.5    0.05       0
Bank Sta=4986.9,5026.5
Exp/Cntr=0.3,0.1

Type RM Length L Ch R = 1,33438,393,393,393
BEGIN DESCRIPTION:
Deadman Creek 30.0
END DESCRIPTION:
XS GIS Cut Line= 3
      1623855.02      6923937.98      1624255.00      6923638.00
      1625410.61      6922484.30
#Sta/Elev= 30
  4499.6 1641.92  4599.6 1638.67  4836.0 1626.19  4863.1 1622.75  4906.9 1612.37
  4921.4 1610.31  4942.3 1603.04  4970.9 1588.66  4972.1 1587.66  5023.8 1588.66
  5027.8 1591.87  5034.9 1594.43  5049.1 1596.69  5119.8 1598.10  5593.5 1595.64
  5869.3 1597.42  5925.9 1594.46  5947.1 1594.99  5954.2 1592.66  5975.4 1592.59
  6053.2 1595.32  6088.5 1594.38  6166.3 1598.03  6350.1 1600.44  6385.5 1603.63
  6420.9 1614.39  6484.5 1627.39  6512.8 1631.59  6555.2 1635.18  6632.5 1636.34
#Mann=3,-1,0
  4499.6    0.05       0  4970.9    0.05       0  5023.8    0.05       0
Bank Sta=4970.9,5023.8
Exp/Cntr=0.3,0.1

Type RM Length L Ch R = 1,33045,1031,1031,1031
BEGIN DESCRIPTION:
Mapping XS d57202fe
END DESCRIPTION:
XS GIS Cut Line= 3
      1624165.16      6924023.27      1624680.81      6923872.22
      1626091.18      6923169.64
#Sta/Elev= 30
  4617.0 1629.29  4741.9 1625.66  4825.2 1616.86  4887.8 1606.63  4908.6 1599.88
  4936.4 1594.16  4941.6 1589.27  4955.4 1587.19  4956.9 1586.19  5021.5 1587.19
  5023.2 1594.28  5033.6 1595.83  5142.2 1596.60  5427.2 1594.85  5488.8 1592.40
  5511.2 1593.82  5550.0 1589.82  5578.3 1596.07  5673.5 1596.47  5684.1 1595.20
  5695.8 1589.69  5785.4 1593.49  5885.2 1592.53  5929.9 1597.08  6367.4 1598.66
  6443.8 1602.76  6456.9 1605.41  6473.7 1612.96  6577.9 1634.99  6730.0 1638.37
#Mann=4,-1,0
  4617.0    0.05       0  4955.4    0.07       0  5021.5    0.05       0
  5142.2    0.05       0
Bank Sta=4955.4,5021.5
Exp/Cntr=0.3,0.1

Type RM Length L Ch R = 1,32014,686,686,686
BEGIN DESCRIPTION:
Deadman Creek 29.0
END DESCRIPTION:
XS GIS Cut Line= 3
      1624255.03      6924088.01      1625155.00      6924388.00
      1626067.03      6924553.07
#Sta/Elev= 30
  4051.6 1626.06  4125.4 1620.01  4188.6 1612.79  4209.7 1608.05  4220.2 1607.54
  4262.4 1597.95  4325.6 1592.84  4568.1 1595.48  4852.7 1593.42  4894.8 1590.66
  4915.9 1591.64  4926.5 1590.57  4947.5 1592.04  4958.1 1590.72  4968.6 1591.09
  4979.2 1589.93  4983.6 1584.79  4984.6 1583.79  5029.1 1583.79  5030.1 1584.79
  5032.1 1584.82  5040.9 1593.05  5051.1 1594.65  5101.9 1592.89  5406.7 1595.08
  5768.1 1601.20  5853.9 1603.01  5869.8 1607.63  5894.5 1612.73  5927.1 1617.76
#Mann=4,-1,0
  4051.6    0.05       0  4983.6    0.05       0  5030.1    0.05       0
  5768.1    0.12       0
Bank Sta=4983.6,5030.1
Exp/Cntr=0.3,0.1

Type RM Length L Ch R = 1,31328,607,607,607
BEGIN DESCRIPTION:
Deadman Creek 28.0
END DESCRIPTION:
XS GIS Cut Line= 3
      1624105.03      6924288.02      1624805.00      6924888.00
      1625768.89      6925320.53
#Sta/Elev= 30
  4083.3 1626.72  4154.1 1624.02  4203.4 1619.27  4217.7 1617.16  4260.5 1607.38
  4289.1 1597.65  4309.9 1594.97  4459.2 1592.58  4537.1 1592.78  4678.7 1589.37
  4750.0 1592.03  4856.5 1591.17  4920.2 1589.26  4969.5 1591.76  4977.2 1590.97
  4982.4 1583.71  4983.4 1582.71  5027.9 1582.71  5028.9 1583.71  5037.2 1589.12
  5042.1 1589.17  5060.0 1589.70  5082.4 1587.96  5125.8 1584.27  5135.4 1585.34
  5147.7 1592.56  5210.4 1591.14  5631.8 1594.79  6042.2 1603.73  6061.7 1605.97
#Mann=5,-1,0
  4083.3    0.05       0  4982.4    0.05       0  5028.9    0.05       0
  5042.1    0.12       0  5082.4    0.05       0
Bank Sta=4982.4,5028.9
Exp/Cntr=0.3,0.1

Type RM Length L Ch R = 1,30721,776,776,776
BEGIN DESCRIPTION:
Deadman Creek 27.0
END DESCRIPTION:
XS GIS Cut Line= 3
      1623800.59      6924840.96      1624956.85      6925601.39
      1626104.98      6925438.00
#Sta/Elev= 30
  4314.7 1627.01  4539.1 1619.21  4575.3 1612.26  4590.3 1603.36  4596.3 1603.64
  4607.4 1598.93  4611.4 1598.96  4626.5 1591.14  4641.6 1589.54  4710.4 1591.19
  4815.7 1590.43  4906.6 1588.82  4915.7 1587.94  4921.8 1584.52  4930.4 1582.21
  4960.7 1581.40  4962.2 1580.40  5027.3 1581.40  5030.1 1583.83  5051.2 1584.79
  5132.6 1584.02  5189.8 1590.90  5397.7 1589.81  5672.5 1599.49  6043.6 1600.29
  6484.6 1608.33  6605.3 1623.04  6706.8 1626.81  6767.4 1632.39  6858.3 1636.94
#Mann=7,-1,0
  4314.7    0.05       0  4607.4    0.12       0  4710.4    0.05       0
  4815.7    0.12       0  4921.8    0.05       0  4960.7    0.05       0
  5027.3    0.05       0
Bank Sta=4960.7,5027.3
Exp/Cntr=0.3,0.1

Type RM Length L Ch R = 1,29945,589,589,589
BEGIN DESCRIPTION:
Deadman Creek 26.0
END DESCRIPTION:
XS GIS Cut Line= 3
      1623754.99      6925237.98      1623955.00      6925738.00
      1625954.99      6925938.00
#Sta/Elev= 30
  4456.2 1622.14  4656.8 1619.10  4818.4 1618.71  4887.0 1613.93  4908.6 1608.15
  4950.3 1601.33  4955.7 1598.07  4979.9 1592.33  4985.3 1587.45  4994.7 1583.78
  4995.8 1578.11  4997.6 1577.11  5075.7 1578.11  5085.2 1584.03  5095.2 1586.30
  5148.0 1588.07  5266.1 1588.11  5316.3 1586.97  5349.0 1582.77  5457.0 1595.09
  5550.0 1598.37  5989.7 1601.82  6311.3 1601.41  6454.5 1603.74  6472.1 1605.41
  6555.0 1607.20  6703.2 1621.71  6833.9 1626.24  6924.3 1631.68  7004.7 1633.29
#Mann=3,-1,0
  4456.2    0.05       0  4995.8    0.05       0  5075.7    0.05       0
Bank Sta=4995.8,5075.7
Exp/Cntr=0.3,0.1

Type RM Length L Ch R = 1,29356,847,847,847
BEGIN DESCRIPTION:
Mapping XS 781b8b91
END DESCRIPTION:
XS GIS Cut Line= 3
      1623472.46      6926200.35      1624071.44      6926278.47
      1625440.57      6926340.94
#Sta/Elev= 30
  4363.7 1618.36  4540.8 1615.95  4598.2 1613.85  4638.5 1609.49  4668.8 1597.00
  4688.7 1585.57  4693.7 1585.10  4699.1 1580.70  4739.4 1584.07  4789.8 1585.29
  4814.5 1584.43  4846.7 1582.77  4870.5 1583.78  4890.7 1579.36  4961.3 1579.62
  4967.0 1579.11  4970.6 1577.11  4971.7 1576.11  5016.2 1576.11  5017.3 1577.11
  5021.4 1585.12  5051.4 1584.29  5061.4 1585.32  5066.7 1587.39  5102.4 1589.38
  5171.5 1592.37  5331.7 1593.60  5652.0 1599.10  6122.5 1600.36  6338.3 1604.11
#Mann=5,-1,0
  4363.7    0.05       0  4814.5    0.12       0  4970.6    0.07       0
  5017.3    0.12       0  5102.4    0.05       0
Bank Sta=4970.6,5017.3
Exp/Cntr=0.3,0.1

Type RM Length L Ch R = 1,28509,716,716,716
BEGIN DESCRIPTION:
Deadman Creek 25.0
END DESCRIPTION:
XS GIS Cut Line= 3
      1623255.01      6926938.00      1623755.00      6926938.00
      1625540.11      6926939.93
#Sta/Elev= 30
  4500.2 1626.15  4700.2 1619.27  4820.2 1609.56  4880.2 1607.15  4900.2 1603.47
  4939.8 1589.19  4970.2 1578.94  4975.0 1572.08  4976.1 1571.08  5020.7 1571.08
  5021.8 1572.08  5030.2 1578.52  5040.2 1582.54  5050.2 1583.93  5064.9 1583.70
  5110.2 1577.10  5120.2 1576.74  5210.2 1580.68  5220.2 1582.09  5240.2 1581.32
  5300.2 1583.25  5320.2 1581.77  5340.2 1582.12  5350.2 1586.34  5400.2 1589.36
  5480.2 1589.57  5710.2 1594.42  6090.2 1595.66  6440.2 1599.37  6785.3 1605.09
#Mann=5,-1,0
  4500.2    0.05       0  4939.8    0.12       0  4975.0    0.07       0
  5021.8    0.12       0  5064.9    0.05       0
Bank Sta=4975,5021.8
Exp/Cntr=0.3,0.1

Type RM Length L Ch R = 1,27793,588,588,588
BEGIN DESCRIPTION:
Deadman Creek 24.0
END DESCRIPTION:
XS GIS Cut Line= 3
      1623352.69      6927627.43      1623705.00      6927638.00
      1625330.95      6927450.45
#Sta/Elev= 30
  4648.0 1622.91  4720.3 1621.01  4810.4 1615.58  4829.6 1609.87  4834.6 1610.51
  4850.4 1604.09  4880.4 1586.16  4890.4 1581.64  4900.4 1580.02  4960.5 1579.90
  4970.0 1571.08  4971.0 1570.08  5015.7 1570.08  5016.7 1571.08  5020.6 1573.04
  5030.7 1575.18  5070.9 1578.27  5081.0 1577.70  5111.2 1579.50  5181.7 1581.72
  5222.8 1581.39  5272.3 1583.87  5332.7 1585.10  5362.9 1587.08  5403.1 1586.82
  5568.5 1590.29  5876.2 1593.13  6003.1 1595.56  6399.7 1596.93  6637.2 1599.28
#Mann=3,-1,0
  4648.0    0.05       0  4970.0    0.05       0  5016.7    0.05       0
Bank Sta=4970,5016.7
Exp/Cntr=0.3,0.1

Type RM Length L Ch R = 1,27205,762,762,762
BEGIN DESCRIPTION:
Deadman Creek 23.0
END DESCRIPTION:
XS GIS Cut Line= 3
      1623254.97      6928087.99      1623765.37      6928181.62
      1625470.15      6927997.60
#Sta/Elev= 30
  4491.2 1613.24  4570.9 1613.85  4576.0 1612.77  4623.4 1614.25  4634.2 1612.86
  4682.3 1613.38  4687.4 1612.33  4775.9 1611.55  4798.7 1610.63  4816.6 1607.88
  4836.9 1606.74  4851.8 1604.76  4887.7 1603.20  4905.0 1591.79  4910.0 1592.97
  4928.4 1580.77  4932.8 1570.85  4934.6 1569.85  5011.2 1569.85  5013.0 1570.85
  5019.8 1570.85  5029.9 1573.07  5039.9 1576.60  5060.0 1579.35  5221.0 1581.28
  5311.5 1583.92  5824.5 1587.50  6176.5 1592.13  6577.6 1594.25  6724.8 1597.52
#Mann=3,-1,0
  4491.2    0.05       0  4932.8    0.03       0  5013.0    0.05       0
Bank Sta=4932.8,5013
Exp/Cntr=0.3,0.1

Type RM Length L Ch R = 1,26443,751,751,751
BEGIN DESCRIPTION:
Deadman Creek 22.0
END DESCRIPTION:
XS GIS Cut Line= 3
      1623205.03      6928788.00      1624004.55      6928853.47
      1625191.19      6928522.25
#Sta/Elev= 30
  4197.8 1611.49  4207.8 1611.27  4256.0 1604.96  4261.0 1605.07  4268.0 1603.51
  4288.1 1601.82  4358.3 1598.61  4388.4 1593.32  4418.5 1590.89  4478.7 1588.58
  4669.3 1583.89  4729.5 1579.99  4769.7 1578.59  4980.4 1577.25  4987.2 1570.38
  4987.9 1569.38  5019.9 1569.38  5020.6 1570.38  5021.2 1571.29  5031.6 1573.04
  5062.8 1573.30  5079.6 1572.45  5116.6 1574.19  5135.8 1577.68  5156.2 1581.49
  5239.3 1583.25  5444.9 1583.28  5613.0 1584.76  5670.7 1586.89  6232.0 1589.02
#Mann=5,-1,0
  4197.8    0.05       0  4987.2    0.03       0  5020.6    0.05       0
  5079.6    0.12       0  5135.8    0.05       0
Bank Sta=4987.2,5020.6
Exp/Cntr=0.3,0.1

Type RM Length L Ch R = 1,25692,1136,1136,1136
BEGIN DESCRIPTION:
Mapping XS ee6747b9
END DESCRIPTION:
XS GIS Cut Line= 4
      1623055.04      6929588.01      1623838.29      6929678.15
      1624570.93      6929372.59      1625700.79      6928268.89
#Sta/Elev= 30
  3748.6 1597.31  3768.7 1594.73  3798.9 1594.47  3859.3 1587.82  4050.1 1584.34
  4292.1 1582.73  4603.1 1583.58  4886.9 1579.81  4934.3 1577.16  4960.2 1569.84
  4961.4 1568.84  5013.8 1569.84  5016.8 1572.71  5022.2 1573.79  5046.0 1575.67
  5162.0 1577.80  5237.7 1578.33  5291.9 1581.11  5506.6 1581.95  5556.2 1585.31
  5626.9 1583.40  5740.1 1583.52  6051.1 1588.09  6631.1 1590.41  6730.1 1591.91
  6779.5 1594.54  6800.8 1593.32  6864.4 1596.79  6885.7 1595.66  6910.3 1599.29
#Mann=4,-1,0
  3748.6    0.05       0  4960.2    0.07       0  5013.8    0.05       0
  5162.0    0.05       0
Bank Sta=4960.2,5013.8
Exp/Cntr=0.3,0.1

Type RM Length L Ch R = 1,24556,446,446,446
BEGIN DESCRIPTION:
Mapping XS 4835d99b
END DESCRIPTION:
XS GIS Cut Line= 4
      1623348.73      6929830.94      1624227.18      6930483.70
      1624897.32      6930497.59      1625605.69      6930445.51
#Sta/Elev= 30
  3430.9 1583.01  3819.3 1580.56  3962.0 1581.13  4055.1 1580.28  4084.3 1581.10
  4169.8 1579.76  4603.2 1578.46  4783.2 1576.86  4813.2 1574.37  4863.2 1573.66
  4923.2 1567.59  4972.9 1566.11  4984.3 1565.91  4985.4 1564.91  5040.2 1564.91
  5041.2 1565.91  5043.3 1567.78  5073.3 1572.30  5179.0 1572.09  5195.6 1571.97
  5213.3 1577.68  5223.4 1579.83  5233.4 1580.38  5464.0 1580.75  5524.2 1581.53
  5530.1 1582.21  5594.4 1583.02  5801.8 1590.75  5806.8 1590.31  5905.9 1592.90
#Mann=5,-1,0
  3430.9    0.05       0  4972.9    0.12       0  4984.3    0.07       0
  5041.2    0.12       0  5179.0    0.05       0
Bank Sta=4984.3,5041.2
Exp/Cntr=0.3,0.1

Type RM Length L Ch R = 1,24110,162,162,162
BEGIN DESCRIPTION:
Mapping XS f7fb606b
END DESCRIPTION:
XS GIS Cut Line= 3
      1622970.19      6930719.81      1624886.90      6930910.79
      1625711.59      6931000.88
#Sta/Elev= 30
  3207.4 1593.80  3704.7 1584.77  3875.5 1586.12  3948.2 1585.55  4116.7 1578.22
  4166.9 1577.53  4207.1 1574.70  4237.3 1576.45  4357.9 1575.95  4378.0 1578.47
  4759.9 1577.13  4870.4 1574.57  4900.6 1568.33  4940.7 1566.95  4968.8 1564.03
  4969.8 1563.03  5024.6 1563.03  5025.7 1564.03  5041.2 1572.75  5114.6 1572.86
  5133.6 1572.28  5141.7 1568.96  5145.4 1568.92  5155.4 1569.58  5182.0 1577.88
  5202.1 1578.94  5443.5 1578.65  5584.4 1579.97  5885.9 1590.72  5963.2 1591.79
#Mann=5,-1,0
  3207.4    0.05       0  4968.8    0.05       0  5025.7    0.05       0
  5114.6    0.12       0  5145.4    0.05       0
Bank Sta=4968.8,5025.7
Exp/Cntr=0.3,0.1

Type RM Length L Ch R = 1,23948,510,510,510
BEGIN DESCRIPTION:
Mapping XS d5fdd162
END DESCRIPTION:
XS GIS Cut Line= 3
      1623046.61      6930869.12      1624616.07      6931046.20
      1625711.69      6931153.69
#Sta/Elev= 30
  3281.5 1593.39  3340.3 1592.59  3380.5 1590.49  3495.4 1589.43  3531.5 1587.68
  3913.9 1583.77  3994.4 1580.70  4085.0 1581.58  4165.5 1576.63  4256.0 1573.58
  4316.4 1576.88  4384.1 1578.44  4799.5 1576.92  4900.0 1573.56  4970.4 1566.46
  4975.9 1563.26  4976.8 1562.26  5023.8 1562.26  5024.7 1563.26  5029.3 1565.01
  5050.8 1564.67  5070.9 1566.13  5090.9 1569.72  5141.2 1575.24  5191.4 1576.94
  5663.7 1578.25  5703.9 1581.94  5844.5 1587.36  5914.9 1587.23  5961.8 1583.90
#Mann=3,-1,0
  3281.5    0.05       0  4975.9    0.03       0  5024.7    0.05       0
Bank Sta=4975.9,5024.7
Exp/Cntr=0.3,0.1

Type RM Length L Ch R = 1,23438,534,534,534
BEGIN DESCRIPTION:
Mapping XS 33f22cfc
END DESCRIPTION:
XS GIS Cut Line= 4
      1624053.54      6931744.13      1624841.76      6931542.73
      1625248.01      6931386.48      1625631.68      6931217.11
#Sta/Elev= 30
  4177.3 1580.93  4223.8 1581.76  4230.4 1582.79  4259.4 1580.54  4300.3 1579.93
  4382.0 1576.09  4447.2 1570.27  4463.6 1570.12  4468.8 1568.00  4488.4 1569.67
  4509.6 1569.37  4571.0 1565.99  4591.7 1572.26  4643.3 1574.61  4785.2 1574.60
  4849.7 1573.31  4901.3 1571.62  4932.3 1569.12  4961.6 1561.22  4962.4 1560.22
  5001.5 1560.22  5002.3 1561.22  5005.0 1564.00  5080.0 1571.82  5108.7 1573.72
  5122.9 1574.81  5431.5 1575.04  5681.0 1577.11  5727.6 1578.16  5845.5 1586.93
#Mann=4,-1,0
  4177.3    0.05       0  4961.6    0.05       0  5002.3    0.05       0
  5108.7    0.05       0
Bank Sta=4961.6,5002.3
Exp/Cntr=0.3,0.1
