HEC-RAS study Long Creek.prj: Long Creek Base Level Engineering

--- Long Creek.g01 (geometry) --- (continued)

Type RM Length L Ch R = 1,67039,462,462,462
BEGIN DESCRIPTION:
Long Creek 110.0
END DESCRIPTION:
XS GIS Cut Line= 3
      1660065.79      6911476.49      1660760.18      6911639.85
      1661030.34      6911670.14
#Sta/Elev= 30
  4291.4 1829.01  4450.3 1826.56  4485.8 1826.48  4582.6 1825.12  4598.8 1824.58
  4681.0 1823.50  4691.2 1823.03  4752.1 1822.38  4783.7 1820.93  4799.6 1822.02
  4896.7 1822.56  4917.2 1823.06  4926.8 1822.75  4948.1 1823.00  4958.3 1822.77
  4968.6 1821.17  4974.3 1819.31  4979.4 1818.94  4989.2 1816.87  4991.6 1815.55
  4992.1 1815.05  5006.7 1815.05  5007.2 1815.55  5009.7 1817.00  5033.9 1817.56
  5039.8 1818.15  5080.0 1819.55  5124.0 1819.78  5160.5 1820.83  5276.6 1821.38
#Mann=3,-1,0
  4291.4    0.05       0  4991.6    0.05       0  5007.2    0.05       0
Bank Sta=4991.6,5007.2
Exp/Cntr=0.3,0.1

Type RM Length L Ch R = 1,66577,485,485,485
BEGIN DESCRIPTION:
Mapping XS 41c04705
END DESCRIPTION:
XS GIS Cut Line= 3
      1660004.98      6911671.78      1660829.67      6912010.34
      1661601.08      6911997.34
#Sta/Elev= 30
  3961.0 1830.47  4018.7 1830.06  4173.3 1826.87  4386.8 1824.20  4624.2 1819.14
  4663.7 1819.82  4778.8 1819.90  4852.5 1819.61  4867.8 1818.89  4947.8 1819.85
  4987.8 1815.35  4988.4 1813.87  4988.9 1813.37  5006.7 1813.37  5007.2 1813.87
  5007.8 1815.00  5047.8 1815.56  5067.8 1815.06  5077.8 1815.72  5097.8 1818.58
  5197.9 1821.28  5285.4 1825.54  5297.9 1825.37  5357.9 1827.50  5467.9 1827.58
  5477.9 1829.70  5507.9 1833.49  5567.9 1838.51  5607.9 1840.51  5624.0 1842.06
#Mann=3,-1,0
  3961.0    0.05       0  4988.4    0.05       0  5007.2    0.05       0
Bank Sta=4988.4,5007.2
Exp/Cntr=0.3,0.1

Type RM Length L Ch R = 1,66092,470,470,470
BEGIN DESCRIPTION:
Long Creek 109.0
END DESCRIPTION:
XS GIS Cut Line= 3
      1659861.75      6911854.06      1660855.00      6912388.00
      1661054.98      6912437.99
#Sta/Elev= 30
  3872.8 1833.19  4062.2 1829.16  4128.0 1828.42  4188.0 1826.98  4335.7 1824.72
  4483.5 1821.56  4631.2 1819.02  4773.2 1817.43  4778.9 1816.66  4839.0 1817.57
  4904.7 1817.02  4910.4 1816.09  4926.6 1814.91  4942.8 1814.90  4955.1 1813.98
  4986.7 1813.11  4988.2 1811.96  4988.7 1811.46  5006.5 1811.46  5007.0 1811.96
  5018.5 1816.37  5031.4 1819.38  5064.9 1823.19  5101.0 1826.40  5106.1 1826.46
  5147.4 1830.71  5175.7 1835.64  5183.4 1838.64  5196.3 1841.12  5206.6 1841.84
#Mann=3,-1,0
  3872.8    0.05       0  4988.2    0.05       0  5007.0    0.05       0
Bank Sta=4988.2,5007
Exp/Cntr=0.3,0.1

Type RM Length L Ch R = 1,65622,404,404,404
BEGIN DESCRIPTION:
Long Creek 108.0
END DESCRIPTION:
XS GIS Cut Line= 3
      1659354.99      6912388.00      1660555.00      6912688.00
      1661004.96      6912688.00
#Sta/Elev= 30
  3758.1 1846.71  3858.6 1840.24  4023.5 1834.13  4193.6 1829.14  4353.4 1826.56
  4366.3 1825.74  4435.8 1824.95  4500.3 1823.23  4675.5 1820.79  4881.7 1815.84
  4964.1 1816.85  4971.8 1815.57  4977.0 1816.38  4992.5 1811.69  4997.5 1811.69
  5005.5 1808.94  5006.0 1808.44  5024.5 1808.94  5025.0 1809.99  5045.0 1812.80
  5055.0 1813.47  5085.0 1813.81  5165.0 1816.56  5245.0 1815.87  5275.0 1817.13
  5365.0 1826.26  5395.0 1830.60  5425.0 1838.13  5435.0 1839.80  5445.0 1840.28
#Mann=3,-1,0
  3758.1    0.05       0  5005.5    0.03       0  5024.5    0.05       0
Bank Sta=5005.5,5024.5
Exp/Cntr=0.3,0.1

Type RM Length L Ch R = 1,65218,167,167,167
BEGIN DESCRIPTION:
Mapping XS 02e9a9a9
END DESCRIPTION:
XS GIS Cut Line= 3
      1659835.75      6913043.32      1660252.42      6913290.72
      1661253.32      6912762.11
#Sta/Elev= 30
  3918.5 1824.51  4301.4 1818.89  4388.3 1816.52  4415.6 1815.97  4437.7 1816.26
  4459.7 1815.47  4620.9 1814.30  4696.2 1815.46  4888.7 1815.08  4903.6 1815.56
  4982.8 1812.14  5015.1 1811.86  5027.6 1810.98  5028.1 1810.48  5046.1 1810.48
  5046.6 1810.98  5081.2 1814.27  5108.8 1817.85  5220.2 1828.08  5310.7 1834.53
  5339.7 1835.01  5345.3 1835.77  5361.7 1835.59  5383.7 1836.76  5422.1 1836.55
  5427.7 1837.55  5444.1 1837.37  5449.8 1838.15  5488.1 1837.90  5535.0 1838.55
#Mann=3,-1,0
  3918.5    0.05       0  5027.6    0.03       0  5046.6    0.05       0
Bank Sta=5027.6,5046.6
Exp/Cntr=0.3,0.1

Type RM Length L Ch R = 1,65051,362,362,362
BEGIN DESCRIPTION:
Mapping XS 3659b328
END DESCRIPTION:
XS GIS Cut Line= 2
      1659853.08      6913668.34      1661467.69      6912839.33
#Sta/Elev= 30
  3826.5 1832.53  3941.1 1827.13  3985.9 1822.71  4008.1 1821.27  4124.7 1816.93
  4141.2 1815.59  4213.4 1815.96  4252.2 1814.84  4363.1 1814.04  4762.5 1814.86
  4862.2 1813.60  4896.6 1813.85  4919.0 1812.09  4964.0 1810.62  4969.3 1809.62
  4969.8 1809.12  4987.8 1809.12  4988.3 1809.62  5039.7 1815.95  5076.4 1818.18
  5084.1 1816.28  5089.7 1818.05  5098.9 1819.51  5150.7 1823.14  5239.4 1826.56
  5366.9 1835.05  5469.4 1839.92  5500.0 1842.09  5527.8 1842.61  5641.5 1847.46
#Mann=4,-1,0
  3826.5    0.05       0  4969.3    0.05       0  4988.3    0.05       0
  5469.4     0.1       0
Bank Sta=4969.3,4988.3
Exp/Cntr=0.3,0.1

Type RM Length L Ch R = 1,64689,471,471,471
BEGIN DESCRIPTION:
Mapping XS 56528d92
END DESCRIPTION:
XS GIS Cut Line= 3
      1659753.33      6913776.82      1660469.43      6913520.75
      1661489.42      6913403.57
#Sta/Elev= 30
  3851.3 1833.09  3952.8 1831.97  4009.1 1828.97  4045.2 1828.06  4108.0 1822.68
  4250.0 1817.19  4275.5 1814.53  4320.4 1815.01  4337.1 1813.56  4362.5 1814.74
  4637.5 1812.87  4889.2 1813.43  4909.3 1812.91  4929.4 1810.99  4969.7 1810.30
  4990.4 1807.93  4990.9 1807.43  5009.4 1807.93  5040.2 1814.50  5050.2 1815.25
  5150.9 1815.11  5332.1 1816.77  5422.7 1818.95  5442.8 1820.28  5462.9 1822.87
  5473.1 1825.71  5533.4 1830.77  5603.9 1834.92  5624.0 1838.42  5638.5 1839.65
#Mann=3,-1,0
  3851.3    0.05       0  4990.4    0.03       0  5009.4    0.05       0
#XS Ineff=2,0
    0.00 4656.70 1819.80               0
Permanent Ineff=
       F       F
Bank Sta=4990.4,5009.4
Exp/Cntr=0.3,0.1

Type RM Length L Ch R = 1,64218,812,812,812
BEGIN DESCRIPTION:
Mapping XS 4f44d4f1
END DESCRIPTION:
XS GIS Cut Line= 3
      1659835.79      6913828.91      1660382.63      6913742.11
      1661510.57      6914245.35
#Sta/Elev= 30
  4090.2 1830.94  4180.5 1827.65  4188.6 1826.69  4193.7 1826.99  4231.2 1822.81
  4250.9 1821.42  4442.8 1814.18  4504.5 1810.14  4545.0 1812.34  4595.7 1812.29
  4657.4 1810.80  4747.4 1812.62  4793.8 1812.70  4822.5 1811.05  4876.4 1811.83
  4938.6 1811.15  4967.3 1810.04  4975.0 1809.21  4982.7 1806.60  4983.2 1806.10
  4999.8 1806.10  5000.3 1806.60  5019.2 1808.81  5037.0 1809.12  5083.4 1812.38
  5140.8 1811.38  5158.6 1812.13  5453.7 1816.05  5799.6 1818.38  5879.0 1820.32
#Mann=3,-1,0
  4090.2    0.05       0  4982.7    0.03       0  5000.3    0.05       0
#XS Ineff=2,0
    0.00 4753.30 1818.24 5246.70    0.00 1818.24
Permanent Ineff=
       F       F
Bank Sta=4982.7,5000.3
Exp/Cntr=0.3,0.1

Type RM Length L Ch R = 1,63406,531,531,531
BEGIN DESCRIPTION:
Mapping XS 8b4583d8
END DESCRIPTION:
XS GIS Cut Line= 2
      1659766.28      6914158.77      1661398.22      6914315.02
#Sta/Elev= 30
  4306.0 1825.16  4425.3 1820.79  4676.4 1815.41  4887.4 1811.91  4917.5 1810.68
  4947.6 1808.82  4957.7 1807.66  4981.3 1807.44  4987.8 1806.78  4997.9 1804.52
  5007.9 1805.75  5018.0 1805.22  5018.2 1803.87  5018.7 1803.37  5037.3 1803.37
  5037.8 1803.87  5038.1 1806.08  5048.1 1808.93  5058.1 1810.22  5098.3 1809.97
  5168.6 1810.73  5228.9 1809.76  5259.1 1810.13  5269.1 1809.58  5294.4 1811.07
  5389.7 1812.79  5660.9 1815.21  5715.2 1815.27  5741.3 1816.05  5945.4 1818.29
#Mann=3,-1,0
  4306.0    0.05       0  5018.2    0.05       0  5037.8    0.05       0
Bank Sta=5018.2,5037.8
Exp/Cntr=0.3,0.1

Type RM Length L Ch R = 1,62875,681,681,681
BEGIN DESCRIPTION:
Long Creek 104.0
END DESCRIPTION:
XS GIS Cut Line= 3
      1659705.01      6914538.00      1660255.00      6914638.00
      1662054.95      6914788.00
#Sta/Elev= 30
  4435.6 1827.85  4506.7 1824.05  4557.6 1818.65  4588.1 1816.99  4914.6 1808.09
  4962.8 1808.22  4967.9 1807.74  4984.4 1803.08  4985.8 1801.71  4986.2 1801.21
  5001.5 1801.71  5024.7 1804.79  5105.0 1808.78  5225.4 1809.01  5235.4 1809.76
  5315.7 1807.65  5345.8 1808.16  5456.2 1804.94  5466.2 1805.37  5496.3 1809.38
  5516.4 1810.34  5827.5 1813.62  6228.9 1821.80  6369.4 1826.43  6376.9 1827.55
  6489.8 1832.50  6539.9 1836.36  6680.4 1841.64  6738.1 1844.95  6800.8 1846.54
#Mann=3,-1,0
  4435.6    0.05       0  4985.8    0.03       0  5001.5    0.05       0
Bank Sta=4985.8,5001.5
Exp/Cntr=0.3,0.1

Type RM Length L Ch R = 1,62194,295,295,295
BEGIN DESCRIPTION:
Mapping XS d4ac7b0f
END DESCRIPTION:
XS GIS Cut Line= 3
      1659691.59      6915086.69      1659938.30      6915151.51
      1661529.73      6915022.98
#Sta/Elev= 30
  4829.8 1813.38  4897.3 1812.64  4926.4 1810.99  4947.1 1806.81  4967.6 1799.09
  4978.1 1797.72  4988.9 1797.33  4989.4 1796.83  5008.1 1796.83  5008.6 1797.33
  5048.3 1799.08  5071.1 1803.35  5080.6 1804.29  5091.6 1804.56  5452.8 1808.16
  5523.0 1807.11  5560.7 1808.14  5693.6 1808.41  5733.7 1807.79  5743.7 1808.18
  5763.8 1807.19  5824.0 1808.78  5914.3 1809.18  6084.8 1811.09  6309.6 1814.66
  6476.1 1818.48  6546.3 1821.08  6554.2 1821.94  6606.5 1823.36  6681.5 1826.30
#Mann=3,-1,0
  4829.8    0.05       0  4988.9    0.03       0  5008.6    0.05       0
Bank Sta=4988.9,5008.6
Exp/Cntr=0.3,0.1

Type RM Length L Ch R = 1,61899,728,728,728
BEGIN DESCRIPTION:
Long Creek 102.0
END DESCRIPTION:
XS GIS Cut Line= 3
      1659654.96      6915388.01      1659905.00      6915338.00
      1661526.90      6915132.17
#Sta/Elev= 30
  4740.2 1816.88  4821.8 1810.41  4842.2 1808.06  4852.4 1805.51  4862.6 1804.73
  4872.8 1802.31  4913.6 1801.17  4954.4 1797.46  4985.0 1797.19  4995.4 1795.95
  4995.9 1795.45  5014.7 1795.45  5015.2 1795.95  5015.3 1796.89  5032.7 1801.72
  5037.7 1801.61  5065.7 1808.22  5085.9 1811.54  5126.2 1805.90  5136.3 1805.61
  5368.2 1806.88  5427.8 1805.07  5569.8 1805.28  5660.5 1808.08  5988.1 1810.56
  6308.2 1815.50  6446.7 1818.44  6527.4 1821.22  6557.6 1822.97  6630.1 1824.49
#Mann=3,-1,0
  4740.2    0.05       0  4995.4    0.05       0  5015.2    0.05       0
Bank Sta=4995.4,5015.2
Exp/Cntr=0.3,0.1

Type RM Length L Ch R = 1,61171,376,376,376
BEGIN DESCRIPTION:
Mapping XS dbdb9eee
END DESCRIPTION:
XS GIS Cut Line= 3
      1659621.28      6916135.82      1660142.15      6915996.93
      1660969.64      6915595.70
#Sta/Elev= 30
  4598.4 1826.13  4613.6 1826.60  4633.3 1824.62  4716.1 1821.81  4728.7 1820.11
  4803.7 1816.85  4829.9 1810.53  4878.8 1806.34  4892.0 1803.88  4912.7 1801.90
  4918.9 1799.90  4943.8 1794.52  4953.8 1793.00  4975.2 1791.64  4975.7 1791.14
  4995.1 1791.64  5039.2 1792.69  5047.3 1795.01  5119.7 1806.80  5136.4 1808.65
  5151.9 1809.33  5162.9 1808.82  5174.5 1805.06  5197.0 1803.03  5685.2 1808.90
  5699.2 1808.47  5970.1 1810.91  6015.2 1811.89  6020.8 1811.24  6057.1 1812.15
#Mann=3,-1,0
  4598.4    0.05       0  4975.2    0.05       0  4995.1    0.05       0
Bank Sta=4975.2,4995.1
Exp/Cntr=0.3,0.1

Type RM Length L Ch R = 1,60795,606,606,606
BEGIN DESCRIPTION:
Long Creek 100.0
END DESCRIPTION:
XS GIS Cut Line= 3
      1659764.03      6916376.69      1660165.67      6916355.94
      1660926.12      6915956.62
#Sta/Elev= 30
  4591.9 1828.46  4602.9 1828.39  4612.9 1827.00  4632.9 1825.96  4642.9 1823.44
  4653.0 1824.05  4683.0 1822.60  4713.0 1822.12  4723.0 1821.13  4733.1 1815.25
  4743.1 1811.55  4783.1 1810.54  4803.2 1807.53  4852.7 1804.56  4933.3 1797.81
  4995.4 1791.40  4995.9 1790.90  5014.8 1790.90  5015.3 1791.40  5043.8 1791.50
  5065.8 1793.14  5104.3 1799.77  5140.2 1808.46  5148.4 1809.72  5162.7 1809.08
  5170.4 1806.13  5185.3 1803.19  5198.1 1803.17  5578.1 1807.79  5853.0 1810.13
#Mann=3,-1,0
  4591.9    0.05       0  4995.4    0.05       0  5015.3    0.05       0
Bank Sta=4995.4,5015.3
Exp/Cntr=0.3,0.1

Type RM Length L Ch R = 1,60189,74,74,74
BEGIN DESCRIPTION:
Long Creek 99.0
END DESCRIPTION:
XS GIS Cut Line= 6
      1659820.90      6916853.23      1660007.08      6916930.38
      1660328.89      6916931.72      1660379.49      6916890.12
      1660308.03      6916388.93      1660943.48      6916008.70
#Sta/Elev= 30
  4599.3 1815.74  4622.4 1816.23  4627.8 1813.45  4646.3 1813.34  4699.5 1804.85
  4722.8 1806.56  4776.5 1798.64  4827.0 1795.98  4838.9 1797.95  4909.3 1790.94
  4909.8 1790.44  4929.2 1790.94  5080.3 1790.94  5110.2 1795.19  5181.6 1796.19
  5242.4 1792.66  5378.9 1795.84  5383.9 1793.71  5423.4 1802.42  5494.3 1805.12
  5524.8 1802.04  5572.6 1802.72  5577.7 1799.71  5625.8 1799.69  5636.6 1796.99
  5684.1 1800.58  5689.1 1798.56  5739.8 1806.60  5804.7 1803.62  6437.2 1809.87
#Mann=3,-1,0
  4599.3    0.05       0  4909.3    0.05       0  4929.2    0.05       0
Bank Sta=4909.3,4929.2
Exp/Cntr=0.3,0.1

Type RM Length L Ch R = 1,60115,81,81,81
BEGIN DESCRIPTION:
Mapping XS b602a746
END DESCRIPTION:
XS GIS Cut Line= 6
      1659792.39      6916878.41      1660163.81      6917014.16
      1660391.41      6916969.24      1660417.65      6916567.93
      1660349.69      6916376.78      1660837.54      6916104.21
#Sta/Elev= 30
  4585.0 1817.29  4588.9 1817.29  4593.6 1815.76  4608.3 1815.58  4658.5 1810.18
  4673.2 1809.48  4679.4 1808.24  4893.1 1809.50  5039.9 1808.35  5127.5 1808.67
  5247.7 1810.69  5255.0 1809.12  5261.0 1810.96  5345.1 1811.37  5390.2 1811.33
  5395.2 1809.58  5445.2 1812.08  5565.3 1812.22  5638.1 1809.58  5654.8 1807.25
  5660.2 1807.69  5685.7 1804.04  5763.0 1802.34  5763.5 1801.84  5782.9 1802.34
  5809.1 1802.46  5815.8 1804.95  5834.6 1806.41  5901.7 1803.74  6397.2 1808.62
#Mann=3,-1,0
  4585.0    0.05       0  5763.0    0.03       0  5782.9    0.05       0
Bank Sta=5763,5782.9
Exp/Cntr=0.3,0.1

Type RM Length L Ch R = 1,60034,120,120,120
BEGIN DESCRIPTION:
Mapping XS 3404a1ed
END DESCRIPTION:
XS GIS Cut Line= 6
      1659773.91      6916880.07      1659918.24      6917023.14
      1660172.79      6917092.02      1660391.41      6917086.03
      1660558.99      6917084.71      1660923.17      6917113.11
#Sta/Elev= 30
  4550.7 1819.40  4557.1 1818.74  4571.2 1814.29  4585.4 1812.34  4592.5 1813.43
  4599.5 1812.28  4606.6 1812.83  4634.9 1810.96  4656.1 1808.56  4663.2 1806.99
  4748.0 1800.02  4771.3 1797.31  4843.8 1793.30  4863.8 1794.31  4869.0 1792.14
  4903.7 1793.96  4908.8 1790.96  4943.5 1792.45  4948.7 1790.47  4968.1 1791.01
  4978.2 1790.55  4978.9 1789.60  4979.4 1789.10  4998.8 1789.60  5119.9 1792.60
  5229.9 1791.30  5420.0 1797.43  5490.2 1798.73  5512.9 1799.97  5769.2 1802.76
#Mann=3,-1,0
  4550.7    0.05       0  4978.9    0.05       0  4998.8    0.05       0
Bank Sta=4978.9,4998.8
Exp/Cntr=0.3,0.1

Type RM Length L Ch R = 1,59914,97,97,97
BEGIN DESCRIPTION:
Mapping XS f8bd76d8
END DESCRIPTION:
XS GIS Cut Line= 5
      1659765.49      6916895.12      1659921.24      6917104.00
      1659981.13      6917160.90      1660457.29      6917271.70
      1660687.88      6917352.56
#Sta/Elev= 30
  4530.6 1817.08  4583.1 1809.87  4603.9 1808.09  4639.4 1807.98  4710.3 1800.84
  4832.0 1797.58  4853.1 1794.46  4883.0 1792.83  5042.1 1791.09  5042.6 1790.59
  5062.4 1791.09  5101.1 1792.56  5113.9 1794.47  5143.7 1792.96  5148.8 1794.40
  5175.5 1793.15  5196.5 1795.13  5216.6 1793.84  5298.7 1795.16  5413.2 1800.60
  5422.8 1799.23  5428.1 1800.55  5445.0 1799.30  5466.2 1801.32  5484.8 1799.57
  5515.8 1799.66  5540.4 1802.22  5546.8 1800.38  5561.6 1799.90  5607.0 1800.21
#Mann=3,-1,0
  4530.6    0.05       0  5042.1    0.03       0  5062.4    0.05       0
Bank Sta=5042.1,5062.4
Exp/Cntr=0.3,0.1

Type RM Length L Ch R = 1,59817,506,506,506
BEGIN DESCRIPTION:
Mapping XS 898a6e31
END DESCRIPTION:
XS GIS Cut Line= 5
      1659735.56      6916978.21      1659879.31      6917208.82
      1660088.94      6917274.70      1660427.34      6917346.57
      1660617.64      6917504.16
#Sta/Elev= 30
  4564.5 1811.35  4623.2 1807.40  4635.2 1805.39  4729.6 1800.03  4854.1 1795.80
  4873.6 1798.02  4886.5 1797.77  4926.1 1794.66  4946.0 1794.74  4957.5 1790.87
  4973.5 1790.33  4974.0 1789.83  4993.8 1790.33  5096.9 1791.75  5113.3 1793.10
  5146.6 1793.37  5191.1 1795.68  5196.2 1794.42  5235.6 1796.01  5240.7 1794.84
  5285.2 1796.13  5290.3 1795.39  5340.0 1795.51  5401.9 1796.48  5443.8 1798.87
  5458.2 1797.96  5479.0 1798.94  5522.0 1799.17  5536.3 1798.43  5649.0 1798.73
#Mann=3,-1,0
  4564.5    0.05       0  4973.5    0.03       0  4993.8    0.05       0
Bank Sta=4973.5,4993.8
Exp/Cntr=0.3,0.1

Type RM Length L Ch R = 1,59311,223,223,223
BEGIN DESCRIPTION:
Mapping XS b6ec2a31
END DESCRIPTION:
XS GIS Cut Line= 3
      1659433.38      6917128.87      1659834.42      6917691.37
      1660370.47      6917930.77
#Sta/Elev= 30
  4310.9 1807.52  4455.6 1804.12  4461.7 1803.89  4476.5 1801.67  4506.0 1800.01
  4648.6 1795.91  4885.8 1795.19  4892.0 1796.07  4899.3 1796.21  4906.7 1795.21
  4936.2 1793.92  4948.5 1791.98  4957.1 1791.58  4963.3 1788.99  4971.9 1787.86
  4978.0 1784.86  4990.4 1781.92  4990.9 1781.42  5014.7 1781.42  5015.2 1781.92
  5024.3 1783.71  5030.0 1786.28  5035.5 1787.64  5068.1 1795.19  5076.4 1796.35
  5111.9 1794.49  5232.3 1796.32  5348.2 1797.12  5573.5 1797.68  5588.8 1797.34
#Mann=3,-1,0
  4310.9    0.05       0  4990.4    0.03       0  5015.2    0.05       0
Bank Sta=4990.4,5015.2
Exp/Cntr=0.3,0.1

Type RM Length L Ch R = 1,59088,181,181,181
BEGIN DESCRIPTION:
Mapping XS 403b7724
END DESCRIPTION:
XS GIS Cut Line= 3
      1659035.44      6917789.53      1660282.34      6917957.00
      1660995.09      6918028.25
#Sta/Elev= 30
  4310.5 1800.81  4330.2 1798.36  4451.3 1795.46  4481.6 1795.37  4491.8 1794.63
  4637.5 1793.51  4743.9 1794.47  4854.9 1794.44  4875.1 1793.29  4925.5 1793.08
  4934.1 1792.65  4945.7 1787.76  4955.8 1785.63  4999.6 1783.95  5000.1 1783.45
  5024.4 1783.95  5026.4 1784.59  5076.9 1787.73  5089.9 1790.64  5097.1 1793.15
  5127.3 1799.78  5157.6 1802.79  5167.8 1801.38  5187.9 1794.86  5198.0 1794.23
  5288.8 1795.52  5882.8 1798.39  5963.2 1799.31  6029.8 1801.17  6284.9 1804.38
#Mann=3,-1,0
  4310.5    0.05       0  4999.6    0.05       0  5024.4    0.05       0
Bank Sta=4999.6,5024.4
Exp/Cntr=0.3,0.1

Type RM Length L Ch R = 1,58907,429,429,429
BEGIN DESCRIPTION:
Mapping XS 7697f69f
END DESCRIPTION:
XS GIS Cut Line= 2
      1658844.81      6917972.62      1660964.59      6918154.91
#Sta/Elev= 30
  4207.7 1808.77  4217.9 1807.64  4288.2 1804.38  4308.3 1802.65  4326.1 1799.34
  4348.4 1797.28  4468.8 1793.89  4519.0 1792.90  4589.3 1792.64  4920.5 1793.59
  4930.5 1792.61  4950.6 1787.16  4960.7 1785.21  4978.4 1783.47  4978.9 1782.97
  5002.7 1782.97  5003.2 1783.47  5051.0 1784.34  5071.1 1785.85  5131.3 1796.00
  5146.1 1797.85  5151.4 1794.12  5161.4 1791.87  5201.5 1791.47  5259.7 1793.12
  5383.3 1794.92  5491.8 1795.80  5763.6 1795.87  5914.2 1797.26  6335.3 1804.28
#Mann=3,-1,0
  4207.7    0.05       0  4978.4    0.03       0  5003.2    0.05       0
Bank Sta=4978.4,5003.2
Exp/Cntr=0.3,0.1

Type RM Length L Ch R = 1,58478,289,289,289
BEGIN DESCRIPTION:
Mapping XS 5d4cdd8c
END DESCRIPTION:
XS GIS Cut Line= 6
      1659104.85      6918056.84      1659449.27      6918090.94
      1659534.53      6918305.80      1659664.13      6918489.97
      1660250.73      6918155.74      1660755.48      6918203.49
#Sta/Elev= 30
  4071.2 1793.49  4151.7 1792.38  4372.8 1792.84  4392.9 1793.67  4412.7 1792.82
  4473.4 1792.55  4586.8 1792.56  4865.8 1791.02  4920.7 1791.34  4933.0 1789.60
  4955.2 1785.03  4964.8 1783.94  4978.2 1781.34  4979.7 1780.29  4980.2 1779.79
  5004.0 1779.79  5004.5 1780.29  5029.6 1785.24  5058.8 1794.98  5067.1 1795.23
  5081.8 1793.90  5094.4 1791.16  5104.5 1790.26  5147.7 1789.56  5250.0 1791.66
  5287.5 1793.70  5346.5 1794.52  5774.1 1796.21  5844.4 1796.96  6055.8 1801.03
#Mann=3,-1,0
  4071.2    0.05       0  4979.7    0.03       0  5004.5    0.05       0
Bank Sta=4979.7,5004.5
Exp/Cntr=0.3,0.1

Type RM Length L Ch R = 1,58189,424,424,424
BEGIN DESCRIPTION:
Mapping XS 882fcac9
END DESCRIPTION:
XS GIS Cut Line= 4
      1659152.61      6918217.03      1659599.69      6918512.19
      1659771.14      6918696.65      1660127.04      6918557.76
#Sta/Elev= 30
  3967.8 1792.54  4092.0 1791.12  4354.0 1791.46  4546.8 1790.21  4582.0 1790.49
  4589.3 1790.06  4610.3 1790.83  4617.7 1790.44  4660.2 1790.96  4849.3 1789.91
  4873.8 1789.17  4879.2 1787.24  4909.8 1783.52  4963.5 1780.08  5013.9 1779.76
  5014.3 1779.26  5035.8 1779.26  5036.3 1779.76  5036.9 1780.31  5042.2 1780.76
  5049.3 1782.67  5060.1 1784.01  5066.7 1785.44  5072.1 1785.77  5091.2 1789.25
  5096.6 1789.38  5121.1 1794.92  5126.4 1794.81  5133.6 1796.16  5137.4 1796.16
#Mann=3,-1,0
  3967.8    0.05       0  5013.9    0.05       0  5036.3    0.05       0
Bank Sta=5013.9,5036.3
Exp/Cntr=0.3,0.1

Type RM Length L Ch R = 1,57765,155,155,155
BEGIN DESCRIPTION:
Long Creek 95.0
END DESCRIPTION:
XS GIS Cut Line= 4
      1659145.78      6918247.85      1659579.75      6918529.53
      1660029.05      6919076.57      1660730.84      6919427.46
#Sta/Elev= 30
  3924.9 1792.69  4098.3 1790.72  4365.1 1791.31  4424.5 1790.27  4452.6 1788.27
  4586.8 1790.03  4615.5 1788.73  4722.4 1788.48  4743.2 1788.69  4757.6 1790.85
  4764.0 1789.56  4786.3 1790.70  4856.6 1788.50  4899.6 1785.38  4920.4 1782.53
  4934.8 1778.87  4943.0 1778.65  4943.5 1778.15  4965.4 1778.65  4984.3 1780.50
  5006.5 1779.43  5020.9 1782.17  5035.2 1779.27  5048.5 1779.15  5062.5 1780.67
  5126.4 1793.12  5201.5 1796.34  5437.4 1799.33  5738.2 1807.12  5934.8 1816.37
#Mann=3,-1,0
  3924.9    0.05       0  4943.0    0.03       0  4965.4    0.05       0
Bank Sta=4943,4965.4
Exp/Cntr=0.3,0.1

Type RM Length L Ch R = 1,57610,241,241,241
BEGIN DESCRIPTION:
Mapping XS 7efccafd
END DESCRIPTION:
XS GIS Cut Line= 3
      1659235.30      6918486.35      1659537.35      6918595.71
      1660058.17      6919470.70
#Sta/Elev= 30
  4142.6 1791.20  4160.2 1791.62  4323.1 1789.51  4364.0 1790.56  4603.1 1789.21
  4630.3 1789.53  4704.4 1789.22  4792.4 1788.47  4799.8 1788.34  4805.6 1787.65
  4836.8 1789.24  4850.5 1788.42  4916.6 1787.24  4966.9 1783.78  4990.2 1783.22
  4999.6 1782.12  5000.1 1781.62  5021.6 1781.62  5022.1 1782.12  5033.5 1782.87
  5039.3 1784.83  5060.7 1788.64  5113.3 1790.88  5214.5 1792.87  5310.0 1793.57
  5325.6 1793.22  5368.4 1794.03  5405.4 1793.58  5448.2 1794.71  5482.1 1794.91
#Mann=3,-1,0
  4142.6    0.05       0  4999.6    0.03       0  5022.1    0.05       0
Bank Sta=4999.6,5022.1
Exp/Cntr=0.3,0.1

Type RM Length L Ch R = 1,57369,566,566,566
BEGIN DESCRIPTION:
Long Creek 94.0
END DESCRIPTION:
XS GIS Cut Line= 3
      1658354.99      6918087.99      1659655.00      6919238.00
      1660455.04      6919888.03
#Sta/Elev= 30
  3286.3 1838.53  3328.5 1836.33  3413.9 1829.07  3491.7 1824.14  3520.1 1820.78
  3654.8 1812.18  3725.9 1805.62  3746.8 1805.21  3810.4 1799.56  3838.8 1795.76
  3881.5 1793.91  4320.6 1788.15  4575.7 1789.70  4724.6 1786.49  4866.0 1786.14
  4880.2 1784.08  4901.8 1783.39  4908.6 1785.96  4915.3 1784.37  4979.7 1783.00
  4996.0 1781.67  4996.5 1781.17  5018.6 1781.67  5035.6 1781.77  5057.9 1786.46
  5121.8 1789.44  5427.1 1792.92  5569.3 1795.74  5889.0 1804.50  6052.8 1814.22
#Mann=3,-1,0
  3286.3    0.05       0  4996.0    0.03       0  5018.6    0.05       0
Bank Sta=4996,5018.6
Exp/Cntr=0.3,0.1

Type RM Length L Ch R = 1,56803,490,490,490
BEGIN DESCRIPTION:
Long Creek 93.0
END DESCRIPTION:
XS GIS Cut Line= 3
      1658454.99      6918737.99      1659205.00      6919538.00
      1660005.02      6920338.02
#Sta/Elev= 30
  3981.3 1808.99  4023.6 1805.41  4242.9 1794.52  4349.4 1794.17  4575.5 1789.71
  4802.2 1782.90  4943.3 1785.10  4957.5 1784.70  4979.0 1780.86  4993.1 1779.86
  4995.2 1778.18  4995.7 1777.68  5017.9 1778.18  5021.5 1779.62  5028.3 1780.01
  5049.8 1779.26  5070.8 1779.93  5074.5 1782.30  5092.0 1784.07  5134.5 1782.77
  5191.0 1783.99  5247.6 1783.31  5304.2 1785.46  5530.5 1785.60  5714.3 1789.04
  5770.9 1789.17  5954.7 1793.62  6082.0 1798.73  6138.6 1802.32  6209.3 1808.42
#Mann=3,-1,0
  3981.3    0.05       0  4995.2    0.03       0  5017.9    0.05       0
Bank Sta=4995.2,5017.9
Exp/Cntr=0.3,0.1

Type RM Length L Ch R = 1,56313,538,538,538
BEGIN DESCRIPTION:
Long Creek 92.0
END DESCRIPTION:
XS GIS Cut Line= 3
      1657954.99      6919287.99      1658755.00      6919738.00
      1660305.04      6920838.03
#Sta/Elev= 30
  4082.5 1822.20  4220.5 1813.05  4449.7 1803.54  4603.6 1794.14  4633.2 1791.11
  4884.1 1784.93  4920.1 1781.77  4933.1 1778.27  4943.0 1777.55  4965.0 1778.72
  4970.8 1778.11  4971.8 1776.89  4972.2 1776.39  4992.1 1776.89  4997.5 1778.69
  5073.0 1782.24  5230.5 1779.57  5280.9 1782.70  5417.3 1783.85  5674.8 1781.86
  5875.1 1785.54  6255.2 1795.91  6377.0 1802.81  6442.2 1809.18  6543.1 1814.01
  6614.4 1821.30  6757.1 1830.77  6778.4 1833.89  6858.0 1839.56  6901.1 1844.19
#Mann=3,-1,0
  4082.5    0.05       0  4971.8    0.05       0  4992.1    0.05       0
Bank Sta=4971.8,4992.1
Exp/Cntr=0.3,0.1

Type RM Length L Ch R = 1,55775,591,591,591
BEGIN DESCRIPTION:
Long Creek 91.0
END DESCRIPTION:
XS GIS Cut Line= 3
      1658055.00      6920038.00      1658505.00      6920188.00
      1660054.98      6920987.99
#Sta/Elev= 30
  4530.3 1800.29  4593.5 1797.86  4656.8 1794.09  4667.3 1792.93  4677.9 1790.32
  4720.0 1783.18  4741.1 1780.85  4899.2 1779.33  4920.3 1778.63  4941.4 1775.71
  4962.5 1775.89  4981.5 1774.72  4982.0 1774.22  5006.8 1774.72  5040.7 1775.63
  5049.7 1777.99  5057.2 1778.92  5190.1 1778.17  5286.0 1780.37  5511.0 1780.77
  5657.3 1778.17  5710.6 1780.36  5865.7 1784.34  6186.3 1791.51  6303.2 1795.33
  6408.3 1800.23  6474.8 1806.23  6629.9 1814.87  6668.6 1820.23  6748.9 1826.65
#Mann=3,-1,0
  4530.3    0.05       0  4981.5    0.03       0  5006.8    0.05       0
Bank Sta=4981.5,5006.8
Exp/Cntr=0.3,0.1

Type RM Length L Ch R = 1,55184,574,574,574
BEGIN DESCRIPTION:
Long Creek 90.0
END DESCRIPTION:
XS GIS Cut Line= 3
      1657705.01      6920688.00      1658505.00      6920738.00
      1660055.03      6921088.01
#Sta/Elev= 30
  4176.9 1810.09  4217.0 1806.16  4317.2 1801.35  4357.2 1797.38  4367.3 1795.67
  4397.3 1786.28  4477.5 1773.18  4497.5 1773.25  4527.6 1775.54  4647.8 1778.26
  4677.9 1777.33  4707.9 1778.85  4808.1 1779.63  4938.4 1776.98  4958.4 1773.92
  4989.9 1771.32  4990.4 1770.82  5015.3 1771.32  5029.7 1773.61  5060.5 1772.40
  5180.6 1777.91  5357.8 1776.08  5419.3 1778.96  5778.1 1785.02  6054.9 1793.25
  6139.1 1796.72  6198.4 1801.25  6403.4 1812.87  6465.0 1819.99  6567.5 1827.93
#Mann=3,-1,0
  4176.9    0.05       0  4989.9    0.03       0  5015.3    0.05       0
Bank Sta=4989.9,5015.3
Exp/Cntr=0.3,0.1

Type RM Length L Ch R = 1,54610,518,518,518
BEGIN DESCRIPTION:
Long Creek 89.0
END DESCRIPTION:
XS GIS Cut Line= 3
      1657605.01      6920838.00      1658405.00      6921288.00
      1659955.02      6921338.00
#Sta/Elev= 30
  4095.5 1814.56  4211.8 1807.59  4227.8 1804.98  4359.4 1799.79  4395.4 1793.96
  4411.3 1788.17  4427.3 1785.64  4462.6 1781.77  4492.3 1776.36  4520.0 1774.47
  4579.0 1773.77  4594.9 1772.29  4713.5 1774.81  4897.0 1773.57  4918.7 1773.04
  4946.1 1769.73  4978.0 1768.87  4982.2 1767.45  4982.6 1766.95  5002.6 1767.45
  5043.4 1769.51  5063.4 1773.72  5083.4 1776.07  5663.7 1780.77  6013.9 1788.27
  6184.0 1794.14  6264.0 1798.23  6404.1 1808.55  6504.1 1814.08  6564.2 1820.88
#Mann=3,-1,0
  4095.5    0.05       0  4982.2    0.03       0  5002.6    0.05       0
Bank Sta=4982.2,5002.6
Exp/Cntr=0.3,0.1

Type RM Length L Ch R = 1,54092,223,223,223
BEGIN DESCRIPTION:
Mapping XS 9d1c1fff
END DESCRIPTION:
XS GIS Cut Line= 3
      1657365.66      6921384.07      1658891.71      6922019.50
      1659407.32      6922035.12
#Sta/Elev= 30
  4241.5 1812.49  4327.4 1808.04  4381.6 1806.36  4520.9 1805.91  4579.5 1803.66
  4609.1 1801.81  4632.5 1797.99  4651.0 1792.54  4656.4 1791.75  4663.2 1788.70
  4680.2 1783.59  4685.6 1783.11  4704.1 1777.65  4709.5 1776.87  4717.4 1772.89
  4733.3 1771.61  4739.1 1770.25  4762.6 1769.53  4887.2 1771.83  4901.6 1770.46
  4916.4 1767.35  4980.6 1767.02  4981.1 1766.52  5006.1 1767.02  5041.1 1767.40
  5070.3 1772.03  5407.3 1774.31  5917.9 1775.91  6158.0 1777.82  6410.4 1783.22
#Mann=3,-1,0
  4241.5    0.05       0  4980.6    0.05       0  5006.1    0.05       0
Bank Sta=4980.6,5006.1
Exp/Cntr=0.3,0.1

Type RM Length L Ch R = 1,53869,497,497,497
BEGIN DESCRIPTION:
Mapping XS c8fcb931
END DESCRIPTION:
XS GIS Cut Line= 4
      1657376.06      6921608.02      1658417.76      6922050.75
      1658896.92      6922201.79      1659301.63      6922310.75
#Sta/Elev= 30
  4371.3 1805.00  4408.9 1802.87  4567.1 1797.58  4685.3 1795.67  4690.8 1795.08
  4714.4 1788.23  4728.7 1785.74  4761.3 1776.92  4767.1 1773.33  4790.8 1767.14
  4814.4 1767.21  4826.5 1769.31  4843.5 1770.35  4925.3 1771.35  4935.2 1771.10
  4949.0 1768.85  4956.9 1766.27  4972.6 1765.36  4979.0 1764.16  4979.5 1763.66
  5002.1 1764.16  5011.2 1766.15  5049.0 1767.39  5096.3 1770.45  5163.3 1769.71
  5201.8 1770.58  5460.0 1771.62  5668.0 1773.81  6129.3 1775.13  6424.7 1777.95
#Mann=3,-1,0
  4371.3    0.05       0  4979.0    0.03       0  5002.1    0.05       0
Bank Sta=4979,5002.1
Exp/Cntr=0.3,0.1

Type RM Length L Ch R = 1,53372,549,549,549
BEGIN DESCRIPTION:
Mapping XS dfdaaa94
END DESCRIPTION:
XS GIS Cut Line= 3
      1657614.01      6922589.89      1658330.16      6922164.54
      1659124.42      6922294.74
#Sta/Elev= 30
  4484.6 1775.89  4537.7 1775.19  4590.3 1773.24  4660.4 1773.34  4829.9 1771.59
  4867.0 1769.50  4888.4 1764.90  4916.1 1765.14  4931.2 1767.18  4952.6 1768.62
  4962.4 1768.37  4968.2 1767.46  4974.2 1765.18  4983.9 1763.45  4987.8 1761.98
  4988.2 1761.48  5008.3 1761.98  5011.1 1764.11  5032.5 1765.79  5122.2 1766.69
  5137.1 1767.53  5165.0 1767.25  5202.1 1769.29  5276.1 1769.33  5430.3 1771.66
  5614.2 1773.18  5864.5 1774.08  5900.1 1775.38  5930.9 1774.48  6122.4 1775.72
#Mann=3,-1,0
  4484.6    0.05       0  4987.8    0.05       0  5008.3    0.05       0
Bank Sta=4987.8,5008.3
Exp/Cntr=0.3,0.1

Type RM Length L Ch R = 1,52823,95,95,95
BEGIN DESCRIPTION:
Mapping XS 40b66b85
END DESCRIPTION:
XS GIS Cut Line= 4
      1657536.91      6922901.95      1658253.58      6922666.14
      1658498.65      6922645.34      1659088.16      6922603.72
#Sta/Elev= 30
  4081.2 1773.48  4089.7 1772.83  4144.7 1773.39  4310.8 1771.69  4437.1 1771.25
  4489.1 1770.40  4500.3 1770.79  4621.6 1768.66  4710.8 1768.38  4780.5 1765.62
  4785.8 1766.12  4805.6 1764.83  4847.1 1765.25  4867.2 1764.65  4877.5 1765.74
  4887.3 1765.65  4907.3 1764.39  4957.5 1763.80  5004.9 1762.04  5005.4 1761.54
  5030.1 1761.54  5030.6 1762.04  5037.8 1763.58  5081.6 1764.68  5098.0 1766.52
  5148.1 1765.76  5218.3 1766.25  5255.1 1768.23  5388.7 1770.60  5672.6 1773.43
#Mann=3,-1,0
  4081.2    0.05       0  5004.9    0.05       0  5030.6    0.05       0
Bank Sta=5004.9,5030.6
Exp/Cntr=0.3,0.1

Type RM Length L Ch R = 1,52728,447,447,447
BEGIN DESCRIPTION:
Mapping XS 9df6a5ec
END DESCRIPTION:
XS GIS Cut Line= 5
      1657694.10      6922999.06      1658230.46      6922767.87
      1658353.00      6922730.88      1658951.80      6922749.37
      1659031.38      6922733.46
#Sta/Elev= 30
  4182.0 1771.15  4449.9 1770.02  4502.3 1770.26  4677.9 1769.17  4753.9 1767.14
  4760.1 1766.38  4765.8 1764.60  4791.7 1764.34  4864.8 1765.40  4875.3 1765.21
  4892.5 1762.87  4936.1 1763.22  4966.9 1762.77  4983.2 1761.95  4983.7 1761.45
  5008.5 1761.45  5009.0 1761.95  5026.1 1762.68  5056.1 1766.73  5106.2 1765.95
  5156.2 1765.85  5166.2 1766.38  5206.2 1766.01  5284.0 1768.29  5289.0 1767.34
  5306.3 1768.64  5356.3 1769.69  5386.3 1768.80  5446.3 1771.00  5574.3 1772.13
#Mann=3,-1,0
  4182.0    0.05       0  4983.2    0.05       0  5009.0    0.05       0
Bank Sta=4983.2,5009
Exp/Cntr=0.3,0.1

Type RM Length L Ch R = 1,52281,230,230,230
BEGIN DESCRIPTION:
Long Creek 86.0
END DESCRIPTION:
XS GIS Cut Line= 3
      1657056.28      6922999.60      1658516.71      6923142.33
      1659558.37      6923276.87
#Sta/Elev= 30
  3582.4 1791.31  3718.4 1780.02  3842.4 1776.26  3993.1 1772.72  4736.6 1767.29
  4817.0 1766.10  4867.2 1763.51  4937.5 1764.69  4967.7 1762.03  4977.7 1759.79
  4979.0 1758.31  4979.4 1757.81  5001.5 1758.31  5038.0 1762.62  5054.1 1761.49
  5078.3 1762.56  5108.6 1760.89  5133.4 1761.38  5148.9 1763.72  5189.2 1765.09
  5259.8 1763.33  5330.4 1765.89  5461.5 1764.14  5520.2 1767.54  5525.2 1766.52
  5592.6 1769.57  5703.5 1776.07  5854.7 1780.37  5945.5 1785.68  6100.1 1790.66
#Mann=3,-1,0
  3582.4    0.05       0  4979.0    0.05       0  5001.5    0.05       0
Bank Sta=4979,5001.5
Exp/Cntr=0.3,0.1

Type RM Length L Ch R = 1,52051,285,285,285
BEGIN DESCRIPTION:
Mapping XS cece27af
END DESCRIPTION:
XS GIS Cut Line= 3
      1657411.42      6923167.97      1658285.19      6923322.29
      1659309.08      6923411.96
#Sta/Elev= 30
  3836.6 1771.74  3850.4 1771.58  3870.7 1769.71  3924.8 1770.83  4114.4 1768.79
  4151.5 1769.12  4165.2 1768.19  4324.0 1767.96  4622.2 1765.05  4713.5 1765.22
  4804.0 1762.27  4874.3 1763.69  4884.3 1763.58  4914.4 1760.51  4954.6 1761.31
  4984.7 1759.82  5014.8 1760.09  5024.8 1761.31  5027.7 1759.42  5028.2 1758.92
  5053.1 1759.42  5065.0 1760.62  5073.0 1762.36  5085.1 1763.19  5215.6 1768.42
  5386.2 1770.74  5607.1 1777.93  5650.6 1780.06  5677.3 1782.32  5751.7 1785.18
#Mann=3,-1,0
  3836.6    0.05       0  5027.7    0.05       0  5053.1    0.05       0
Bank Sta=5027.7,5053.1
Exp/Cntr=0.3,0.1

Type RM Length L Ch R = 1,51766,477,477,477
BEGIN DESCRIPTION:
Long Creek 85.0
END DESCRIPTION:
XS GIS Cut Line= 3
      1656936.89      6923081.57      1658555.00      6923588.00
      1658954.99      6923937.99
#Sta/Elev= 30
  3302.1 1799.97  3338.6 1795.77  3441.2 1788.47  3506.1 1781.30  3635.4 1773.46
  3641.2 1774.87  3646.4 1773.79  3666.9 1774.48  3761.2 1772.23  3824.0 1768.60
  3865.9 1770.32  4096.5 1767.13  4748.9 1763.32  4813.9 1761.54  4840.4 1762.30
  4916.5 1758.56  4943.7 1761.22  4992.5 1754.56  4992.9 1754.06  5015.0 1754.56
  5033.2 1755.81  5054.1 1761.69  5082.6 1767.62  5090.1 1767.97  5096.8 1764.77
  5111.0 1762.49  5266.7 1762.84  5401.5 1772.16  5458.4 1778.29  5529.1 1781.85
#Mann=3,-1,0
  3302.1    0.05       0  4992.5    0.03       0  5015.0    0.05       0
Bank Sta=4992.5,5015
Exp/Cntr=0.3,0.1

Type RM Length L Ch R = 1,51289,471,471,471
BEGIN DESCRIPTION:
Long Creek 84.0
END DESCRIPTION:
XS GIS Cut Line= 3
      1656755.00      6923238.00      1658205.00      6923938.00
      1658855.00      6924088.00
#Sta/Elev= 30
  3346.1 1814.49  3473.2 1807.94  3518.4 1802.06  3682.2 1785.89  3757.0 1775.31
  3801.4 1771.72  3981.6 1766.93  4004.2 1765.03  4049.4 1766.27  4223.3 1763.85
  4557.9 1762.97  4670.9 1760.40  4925.1 1761.15  4934.0 1760.98  4953.4 1754.94
  4978.3 1750.23  4978.7 1749.73  5000.9 1750.23  5065.7 1761.90  5108.5 1767.53
  5120.4 1763.03  5130.7 1761.45  5253.8 1762.39  5284.6 1760.92  5305.2 1757.54
  5325.7 1757.14  5380.4 1762.46  5407.8 1762.66  5551.5 1776.72  5623.3 1780.73
#Mann=3,-1,0
  3346.1    0.05       0  4978.3    0.03       0  5000.9    0.05       0
Bank Sta=4978.3,5000.9
Exp/Cntr=0.3,0.1

Type RM Length L Ch R = 1,50818,309,309,309
BEGIN DESCRIPTION:
Long Creek 83.0
END DESCRIPTION:
XS GIS Cut Line= 4
      1657191.74      6923491.81      1657842.75      6923822.52
      1658097.96      6924593.36      1658754.98      6924987.99
#Sta/Elev= 30
  3707.0 1770.00  3846.5 1766.42  3863.1 1764.36  3923.8 1765.69  4069.6 1764.22
  4080.1 1763.43  4092.0 1764.21  4338.8 1763.10  4428.5 1762.08  4528.2 1759.32
  4655.0 1760.13  4744.9 1758.22  4781.9 1758.82  4801.1 1757.36  4822.2 1757.05
  4877.0 1759.84  4895.9 1759.94  4966.9 1755.23  4984.4 1752.90  4984.9 1752.40
  5012.7 1752.90  5035.5 1754.89  5053.9 1755.08  5075.0 1760.09  5085.5 1760.90
  5329.7 1759.40  5541.5 1761.64  5737.8 1766.90  5885.4 1773.98  6015.6 1778.88
#Mann=3,-1,0
  3707.0    0.05       0  4984.4    0.03       0  5012.7    0.05       0
Bank Sta=4984.4,5012.7
Exp/Cntr=0.3,0.1

Type RM Length L Ch R = 1,50509,484,484,484
BEGIN DESCRIPTION:
Mapping XS 14d1f56f
END DESCRIPTION:
XS GIS Cut Line= 4
      1657603.29      6923783.14      1657763.86      6924573.47
      1657986.99      6924688.17      1658460.63      6924931.62
#Sta/Elev= 30
  4313.2 1762.89  4542.7 1761.52  4649.0 1756.83  4654.9 1754.79  4675.3 1752.34
  4699.6 1756.49  4726.3 1755.22  4777.3 1755.82  4795.8 1754.89  4910.0 1757.16
  4930.4 1756.04  4947.7 1751.88  4952.8 1753.12  4973.8 1749.81  4974.2 1749.31
  4996.5 1749.81  5012.0 1751.56  5042.7 1759.30  5048.9 1762.00  5054.0 1761.97
  5063.1 1763.93  5083.5 1762.43  5093.7 1759.62  5099.5 1759.24  5383.2 1758.78
  5427.5 1756.94  5480.8 1758.88  5525.7 1758.66  5749.0 1761.70  5903.1 1765.44
#Mann=3,-1,0
  4313.2    0.05       0  4973.8    0.05       0  4996.5    0.05       0
Bank Sta=4973.8,4996.5
Exp/Cntr=0.3,0.1

Type RM Length L Ch R = 1,50025,627,627,627
BEGIN DESCRIPTION:
Long Creek 82.0
END DESCRIPTION:
XS GIS Cut Line= 4
      1656754.99      6924037.99      1657373.33      6924369.28
      1657980.05      6924705.08      1658434.01      6924956.33
#Sta/Elev= 30
  4298.5 1810.83  4363.6 1801.95  4416.3 1795.35  4438.2 1788.83  4454.5 1781.40
  4476.4 1775.92  4521.8 1768.71  4570.8 1762.18  4651.9 1759.41  4763.7 1758.40
  4837.9 1755.83  4911.1 1757.93  4925.7 1753.15  4981.8 1747.72  4982.2 1747.22
  5004.6 1747.72  5013.4 1751.48  5051.2 1759.20  5067.2 1758.21  5072.9 1755.33
  5081.9 1755.44  5089.0 1758.00  5094.7 1756.08  5116.4 1755.96  5398.1 1759.19
  5685.6 1758.62  5750.8 1756.82  5788.6 1758.67  6081.8 1761.69  6212.3 1764.84
#Mann=5,-1,0
  4298.5    0.05       0  4363.6    0.12       0  4521.8    0.05       0
  4981.8    0.03       0  5004.6    0.05       0
Bank Sta=4981.8,5004.6
Exp/Cntr=0.3,0.1

Type RM Length L Ch R = 1,49398,260,260,260
BEGIN DESCRIPTION:
Long Creek 81.0
END DESCRIPTION:
XS GIS Cut Line= 3
      1656709.97      6924340.79      1657142.23      6924872.00
      1658255.02      6926088.02
#Sta/Elev= 30
  4272.8 1803.20  4331.7 1796.21  4352.5 1790.19  4381.3 1785.00  4387.7 1781.55
  4402.1 1777.75  4480.4 1766.71  4544.3 1760.02  4694.4 1754.15  4907.0 1752.91
  4942.2 1751.12  4978.3 1743.83  4992.2 1742.64  4992.7 1742.14  5020.8 1742.64
  5056.0 1752.06  5098.5 1755.85  5119.5 1760.78  5126.9 1760.39  5133.7 1762.73
  5141.1 1761.80  5147.9 1763.89  5155.3 1761.53  5162.0 1762.94  5176.2 1756.60
  5353.2 1759.94  5841.6 1763.42  6202.4 1773.26  6478.6 1788.08  6606.0 1789.43
#Mann=3,-1,0
  4272.8    0.05       0  4992.2    0.05       0  5020.8    0.05       0
Bank Sta=4992.2,5020.8
Exp/Cntr=0.3,0.1

Type RM Length L Ch R = 1,49138,229,229,229
BEGIN DESCRIPTION:
Mapping XS 656c127c
END DESCRIPTION:
XS GIS Cut Line= 5
      1656664.90      6924492.14      1656900.55      6924713.19
      1656998.55      6924888.36      1657100.73      6925126.08
      1657540.37      6925532.37
#Sta/Elev= 30
  4548.9 1800.66  4595.5 1794.03  4666.3 1774.11  4772.3 1759.11  4923.4 1752.37
  4968.4 1754.12  4998.0 1750.29  4998.4 1749.79  5020.9 1750.29  5033.5 1757.49
  5049.4 1759.06  5055.2 1756.55  5060.9 1758.23  5069.7 1756.37  5077.1 1759.09
  5100.6 1756.60  5106.1 1759.29  5159.4 1758.71  5176.7 1755.73  5182.2 1758.95
  5200.3 1756.43  5205.7 1759.56  5223.8 1756.19  5229.2 1759.33  5252.8 1754.40
  5258.2 1757.16  5276.3 1755.36  5281.8 1757.59  5299.9 1754.41  5930.1 1760.78
#Mann=3,-1,0
  4548.9    0.05       0  4998.0    0.03       0  5020.9    0.05       0
Bank Sta=4998,5020.9
Exp/Cntr=0.3,0.1

Type RM Length L Ch R = 1,48909,557,557,557
BEGIN DESCRIPTION:
Long Creek 80.0
END DESCRIPTION:
XS GIS Cut Line= 3
      1656504.97      6924737.98      1656955.00      6925088.00
      1658055.02      6926038.02
#Sta/Elev= 30
  4529.4 1802.36  4580.7 1795.87  4629.9 1787.12  4679.7 1772.99  4764.7 1758.29
  4793.7 1754.97  4808.1 1751.70  4820.8 1750.82  4849.8 1753.16  4878.7 1750.65
  4922.2 1749.33  4963.8 1752.83  4978.3 1751.05  4992.7 1746.72  5028.0 1747.78
  5057.1 1746.05  5057.6 1745.55  5085.8 1746.05  5120.9 1746.47  5170.3 1752.08
  5198.8 1753.77  5241.6 1754.35  5248.2 1752.49  5262.4 1751.29  5297.7 1755.18
  5390.2 1757.92  5851.5 1760.34  6127.9 1765.27  6283.7 1770.44  6553.0 1787.22
#Mann=4,-1,0
  4529.4    0.12       0  4580.7    0.05       0  5057.1    0.03       0
  5085.8    0.05       0
Bank Sta=5057.1,5085.8
Exp/Cntr=0.3,0.1

Type RM Length L Ch R = 1,48352,271,271,271
BEGIN DESCRIPTION:
Long Creek 79.0
END DESCRIPTION:
XS GIS Cut Line= 3
      1656405.02      6924988.04      1656555.00      6925388.00
      1657227.62      6925983.49
#Sta/Elev= 30
  4567.6 1790.29  4588.9 1786.67  4607.6 1785.79  4662.8 1779.96  4698.4 1770.49
  4723.3 1765.80  4728.6 1763.58  4748.2 1762.20  4791.8 1755.79  4808.7 1754.54
  4814.1 1753.37  4863.9 1750.82  4894.2 1747.28  4962.7 1747.76  4985.0 1745.96
  4987.5 1744.31  4988.0 1743.81  5016.2 1744.31  5022.8 1746.40  5030.3 1746.55
  5051.2 1750.41  5058.7 1750.57  5122.3 1749.49  5143.2 1748.01  5171.6 1751.59
  5214.3 1752.73  5773.9 1756.78  5781.4 1756.06  5795.6 1756.88  5893.1 1757.76
#Mann=3,-1,0
  4567.6    0.05       0  4987.5    0.03       0  5016.2    0.05       0
Bank Sta=4987.5,5016.2
Exp/Cntr=0.3,0.1

Type RM Length L Ch R = 1,48081,293,293,293
BEGIN DESCRIPTION:
Mapping XS e8409ba4
END DESCRIPTION:
XS GIS Cut Line= 2
      1656149.84      6925342.95      1656648.21      6925889.29
#Sta/Elev= 30
  4680.7 1770.29  4687.6 1768.65  4695.0 1765.64  4701.8 1765.48  4709.2 1763.30
  4744.4 1759.39  4751.8 1756.62  4758.6 1756.58  4780.2 1753.99  4794.3 1753.17
  4815.3 1750.51  4843.7 1748.60  4857.9 1748.90  4886.2 1746.18  4921.4 1746.34
  4949.8 1744.72  4971.0 1744.51  4971.5 1744.01  4999.2 1744.01  4999.7 1744.51
  5013.3 1746.89  5027.5 1747.59  5055.8 1746.91  5077.4 1747.59  5084.2 1748.81
  5098.4 1749.53  5147.7 1751.11  5190.3 1751.04  5240.3 1751.92  5420.2 1753.21
#Mann=3,-1,0
  4680.7    0.05       0  4971.0    0.05       0  4999.7    0.05       0
Bank Sta=4971,4999.7
Exp/Cntr=0.3,0.1

Type RM Length L Ch R = 1,47788,502,502,502
BEGIN DESCRIPTION:
Long Creek 78.0
END DESCRIPTION:
XS GIS Cut Line= 3
      1655897.49      6925336.66      1656155.00      6925788.00
      1656630.00      6926063.00
#Sta/Elev= 30
  4494.7 1773.11  4507.8 1772.15  4516.7 1768.90  4522.5 1768.60  4559.9 1761.96
  4581.5 1760.47  4603.1 1758.14  4619.0 1755.54  4646.3 1753.87  4668.9 1751.23
  4699.6 1749.61  4807.7 1747.39  4830.1 1747.53  4853.2 1746.05  4941.6 1744.96
  4956.8 1743.75  4963.2 1742.48  4986.3 1741.94  4986.8 1741.44  5014.5 1741.44
  5015.0 1741.94  5022.2 1742.75  5043.7 1747.90  5059.5 1749.17  5118.3 1749.78
  5129.9 1749.07  5145.6 1749.75  5153.0 1749.26  5167.2 1750.59  5563.2 1754.21
#Mann=3,-1,0
  4494.7    0.05       0  4986.3    0.05       0  5015.0    0.05       0
Bank Sta=4986.3,5015
Exp/Cntr=0.3,0.1

Type RM Length L Ch R = 1,47286,315,315,315
BEGIN DESCRIPTION:
Long Creek 77.0
END DESCRIPTION:
XS GIS Cut Line= 3
      1655655.00      6925337.98      1655705.00      6925938.00
      1655763.76      6926907.62
#Sta/Elev= 30
  4379.8 1778.97  4409.9 1776.58  4430.0 1773.21  4437.5 1769.18  4442.5 1768.89
  4450.1 1766.03  4470.1 1762.18  4557.9 1751.66  4610.6 1748.54  4670.8 1747.07
  4841.4 1746.47  4851.4 1748.01  4891.6 1746.04  4919.2 1742.89  4971.9 1742.95
  4984.4 1741.97  4987.5 1740.42  4988.0 1739.92  5016.3 1740.42  5032.0 1742.56
  5052.0 1746.52  5122.2 1745.77  5152.2 1743.26  5202.3 1743.21  5222.3 1744.70
  5228.6 1746.47  5233.6 1744.54  5252.4 1747.55  5312.5 1750.22  5953.3 1758.68
#Mann=3,-1,0
  4379.8    0.05       0  4987.5    0.03       0  5016.3    0.05       0
Bank Sta=4987.5,5016.3
Exp/Cntr=0.3,0.1

Type RM Length L Ch R = 1,46971,67,67,67
BEGIN DESCRIPTION:
Mapping XS 6a6598b4
END DESCRIPTION:
XS GIS Cut Line= 6
      1655575.76      6925302.59      1655396.06      6925961.46
      1655406.48      6926031.78      1655437.73      6926081.26
      1655531.48      6926109.90      1655471.58      6927010.93
#Sta/Elev= 30
  4392.3 1779.63  4471.1 1773.84  4484.1 1771.95  4511.8 1762.34  4523.3 1760.57
  4616.0 1750.60  4654.2 1748.25  4784.4 1747.17  4815.8 1751.27  4864.3 1751.05
  4869.4 1753.19  4913.7 1751.14  4918.8 1753.54  4958.0 1751.77  4969.9 1753.35
  5007.5 1751.37  5166.0 1751.38  5172.0 1749.41  5177.9 1750.52  5187.3 1747.58
  5193.2 1749.82  5202.7 1743.97  5203.2 1743.47  5232.8 1743.97  5232.9 1746.21
  5273.3 1750.19  5415.0 1746.05  5445.1 1748.24  5525.3 1747.72  6209.7 1760.87
#Mann=3,-1,0
  4392.3    0.05       0  5202.7    0.03       0  5232.8    0.05       0
Bank Sta=5202.7,5232.8
Exp/Cntr=0.3,0.1

Type RM Length L Ch R = 1,46904,377,377,377
BEGIN DESCRIPTION:
Mapping XS 5c044ec4
END DESCRIPTION:
XS GIS Cut Line= 5
      1655475.60      6925257.34      1655344.64      6925644.23
      1655344.64      6926033.21      1655433.18      6926309.25
      1655344.92      6926714.22
#Sta/Elev= 30
  4348.8 1778.49  4391.7 1775.74  4402.5 1774.04  4428.7 1772.20  4476.2 1762.18
  4539.5 1755.60  4560.6 1752.34  4634.5 1747.62  4711.5 1746.29  4851.0 1747.02
  4901.0 1744.95  4921.0 1740.57  4961.0 1742.19  5041.0 1740.81  5071.0 1742.79
  5111.0 1743.02  5146.1 1745.56  5245.8 1745.17  5252.0 1740.43  5252.5 1739.93
  5282.1 1740.43  5293.9 1742.46  5319.3 1741.04  5326.0 1744.74  5331.3 1743.41
  5350.8 1745.82  5436.1 1746.66  5685.7 1752.68  5721.4 1752.42  5850.6 1754.61
#Mann=3,-1,0
  4348.8    0.05       0  5252.0    0.03       0  5282.1    0.05       0
Bank Sta=5252,5282.1
Exp/Cntr=0.3,0.1

Type RM Length L Ch R = 1,46527,497,497,497
BEGIN DESCRIPTION:
Mapping XS 50a30775
END DESCRIPTION:
XS GIS Cut Line= 2
      1655032.14      6925184.29      1654933.18      6926699.86
#Sta/Elev= 30
  4327.5 1767.56  4331.8 1767.56  4351.3 1763.06  4371.3 1760.21  4441.5 1754.82
  4491.6 1747.59  4510.2 1746.60  4551.7 1745.01  4862.3 1745.43  4952.5 1744.81
  4962.6 1743.33  4970.9 1740.22  4975.9 1741.15  4987.6 1736.44  4988.1 1735.94
  5017.7 1736.44  5032.7 1737.62  5072.8 1744.64  5082.8 1745.40  5092.8 1745.54
  5112.9 1742.58  5163.0 1744.16  5293.3 1743.52  5313.3 1742.77  5333.3 1739.46
  5343.4 1739.04  5373.4 1743.56  5436.6 1746.88  5664.0 1750.96  5846.3 1755.79
#Mann=3,-1,0
  4327.5    0.05       0  4987.6    0.03       0  5017.7    0.05       0
Bank Sta=4987.6,5017.7
Exp/Cntr=0.3,0.1

Type RM Length L Ch R = 1,46030,318,318,318
BEGIN DESCRIPTION:
Mapping XS 615f0f30
END DESCRIPTION:
XS GIS Cut Line= 6
      1654946.61      6925307.52      1654892.39      6925695.37
      1654448.22      6925749.59      1654441.97      6926076.98
      1654667.18      6926237.55      1654650.59      6926484.33
#Sta/Elev= 30
  4309.3 1748.32  4356.1 1745.04  4722.4 1743.82  4762.8 1757.97  4886.2 1750.11
  5146.5 1747.10  5171.8 1744.15  5176.7 1740.55  5177.2 1740.05  5206.9 1740.55
  5271.9 1748.03  5322.0 1745.93  5452.1 1750.23  5486.0 1743.75  5520.7 1746.69
  5526.8 1744.25  5541.6 1748.39  5547.7 1745.16  5562.5 1744.32  5577.2 1747.84
  5598.1 1744.63  5627.6 1748.26  5648.5 1745.42  5663.3 1748.51  5669.4 1745.80
  5684.2 1749.88  5734.6 1752.49  5768.1 1751.39  5798.2 1746.11  6005.0 1750.95
#Mann=3,-1,0
  4309.3    0.05       0  5176.7    0.03       0  5206.9    0.05       0
Bank Sta=5176.7,5206.9
Exp/Cntr=0.3,0.1

Type RM Length L Ch R = 1,45712,492,492,492
BEGIN DESCRIPTION:
Long Creek 74.0
END DESCRIPTION:
XS GIS Cut Line= 3
      1654965.18      6924977.01      1654465.15      6925459.67
      1654086.66      6926261.78
#Sta/Elev= 30
  4291.8 1775.55  4328.0 1773.29  4384.6 1768.27  4441.2 1761.00  4476.4 1759.44
  4526.1 1754.48  4540.2 1753.83  4561.3 1749.49  4575.5 1747.88  4582.7 1748.09
  4611.0 1745.79  4752.2 1742.42  4950.3 1741.58  4964.5 1738.98  4978.6 1734.24
  4979.5 1733.30  4980.0 1732.80  5009.7 1733.30  5029.2 1737.70  5068.5 1740.37
  5142.4 1740.63  5205.1 1739.66  5227.9 1741.41  5279.0 1742.16  5427.2 1741.18
  5615.2 1741.52  5758.9 1744.26  5819.4 1749.63  5858.5 1758.04  5873.7 1759.36
#Mann=3,-1,0
  4291.8    0.05       0  4979.5    0.03       0  5009.7    0.05       0
Bank Sta=4979.5,5009.7
Exp/Cntr=0.3,0.1

Type RM Length L Ch R = 1,45220,500,500,500
BEGIN DESCRIPTION:
Long Creek 73.0
END DESCRIPTION:
XS GIS Cut Line= 3
      1654306.60      6924968.63      1654020.22      6925338.52
      1653968.08      6926113.77
#Sta/Elev= 30
  4532.2 1748.64  4632.6 1747.48  4783.0 1744.53  4903.4 1743.21  4938.7 1739.78
  4946.9 1737.05  4953.2 1737.87  4961.4 1736.33  4967.7 1736.48  4981.4 1734.47
  4981.9 1733.97  5011.1 1733.97  5011.6 1734.47  5049.6 1734.75  5069.6 1737.40
  5079.7 1737.52  5099.7 1739.11  5109.7 1739.32  5148.5 1738.21  5159.8 1738.28
  5189.9 1739.84  5240.0 1740.26  5610.9 1739.40  5671.0 1739.65  5691.0 1740.04
  5741.1 1742.80  5747.3 1743.98  5761.2 1744.73  5771.2 1746.01  5777.0 1747.33
#Mann=3,-1,0
  4532.2    0.05       0  4981.4    0.03       0  5011.6    0.05       0
Bank Sta=4981.4,5011.6
Exp/Cntr=0.3,0.1

Type RM Length L Ch R = 1,44720,458,458,458
BEGIN DESCRIPTION:
Long Creek 72.0
END DESCRIPTION:
XS GIS Cut Line= 3
      1653568.38      6924520.35      1653539.81      6925337.47
      1653658.64      6926041.09
#Sta/Elev= 30
  4171.4 1753.35  4199.4 1751.01  4229.1 1748.70  4289.1 1747.08  4429.2 1744.50
  4555.5 1743.43  4929.5 1740.66  4949.5 1739.37  4959.5 1737.40  4979.1 1731.24
  4984.1 1732.59  4984.5 1730.82  4985.0 1730.32  5014.9 1730.82  5020.0 1732.44
  5070.7 1736.05  5192.4 1737.72  5385.1 1738.24  5526.3 1736.33  5531.4 1737.14
  5547.3 1737.03  5567.6 1738.48  5586.8 1741.86  5591.8 1740.63  5638.6 1753.78
  5647.2 1757.22  5652.3 1754.71  5658.9 1757.43  5669.0 1758.45  5702.6 1758.41
#Mann=5,-1,0
  4171.4    0.05       0  4199.4    0.12       0  4555.5    0.05       0
  4984.5    0.05       0  5014.9    0.05       0
Bank Sta=4984.5,5014.9
Exp/Cntr=0.3,0.1
