HEC-RAS study Long Creek.prj: Long Creek Base Level Engineering

--- Long Creek.g01 (geometry) --- (continued)

Type RM Length L Ch R = 1,44262,56,56,56
BEGIN DESCRIPTION:
Mapping XS 435a6554
END DESCRIPTION:
XS GIS Cut Line= 5
      1653253.22      6924716.39      1653226.23      6925042.67
      1653180.36      6925597.36      1653211.64      6925732.90
      1653349.29      6925901.84
#Sta/Elev= 30
  4083.3 1742.20  4586.6 1738.22  4646.8 1737.02  4717.1 1737.49  4730.5 1736.56
  4767.2 1746.19  4787.3 1746.63  4807.4 1745.54  4846.4 1740.56  4851.4 1738.40
  4857.5 1737.05  4907.7 1734.26  4965.1 1727.47  4996.9 1726.23  4997.4 1725.73
  5027.4 1726.23  5049.8 1730.36  5054.9 1730.62  5060.3 1734.31  5091.1 1741.93
  5097.7 1744.64  5106.4 1744.74  5119.5 1749.40  5133.9 1751.93  5140.3 1750.10
  5148.2 1751.13  5154.7 1749.08  5240.9 1750.86  5247.3 1751.60  5324.3 1752.38
#Mann=3,-1,0
  4083.3    0.05       0  4996.9    0.05       0  5027.4    0.05       0
Bank Sta=4996.9,5027.4
Exp/Cntr=0.3,0.1

Type RM Length L Ch R = 1,44206,191,191,191
BEGIN DESCRIPTION:
Mapping XS 75ef4cda
END DESCRIPTION:
XS GIS Cut Line= 4
      1653194.95      6924988.46      1653138.65      6925507.69
      1653130.31      6925624.47      1653188.70      6925858.03
#Sta/Elev= 30
  4327.1 1739.47  4407.1 1739.25  4658.6 1736.53  4835.7 1736.69  4884.6 1735.19
  4885.1 1734.69  4914.6 1734.69  4915.1 1735.19  4919.9 1737.74  4949.9 1740.59
  4960.0 1740.57  4965.7 1741.12  5006.3 1740.00  5011.4 1740.55  5031.9 1740.67
  5042.2 1740.14  5047.5 1739.25  5052.7 1740.99  5073.2 1742.05  5088.8 1741.36
  5093.9 1742.18  5130.0 1741.45  5135.1 1743.25  5155.6 1742.46  5165.9 1743.80
  5171.2 1747.42  5176.4 1748.10  5186.6 1752.02  5196.9 1753.80  5207.2 1753.21
#Mann=3,-1,0
  4327.1    0.05       0  4884.6    0.05       0  4915.1    0.05       0
Bank Sta=4884.6,4915.1
Exp/Cntr=0.3,0.1

Type RM Length L Ch R = 1,44015,545,545,545
BEGIN DESCRIPTION:
Long Creek 71.0
END DESCRIPTION:
XS GIS Cut Line= 3
      1653089.75      6924476.59      1652955.00      6925738.00
      1652905.00      6926138.00
#Sta/Elev= 30
  3757.4 1751.82  3809.1 1746.12  3839.3 1743.71  3909.7 1741.16  4070.6 1739.12
  4342.1 1737.60  4462.8 1735.72  4593.5 1735.48  4774.6 1736.88  4855.0 1735.83
  4875.1 1738.50  4882.5 1737.27  4887.5 1737.78  4895.2 1735.69  4905.3 1734.39
  4970.3 1729.37  4970.8 1728.87  5001.3 1729.37  5036.1 1730.38  5063.8 1738.39
  5076.4 1740.40  5144.4 1743.49  5157.0 1745.17  5217.5 1750.21  5225.0 1751.78
  5230.1 1751.64  5247.7 1754.88  5277.9 1754.52  5305.6 1756.56  5429.1 1759.67
#Mann=3,-1,0
  3757.4    0.05       0  4970.3    0.05       0  5001.3    0.05       0
Bank Sta=4970.3,5001.3
Exp/Cntr=0.3,0.1

Type RM Length L Ch R = 1,43470,599,599,599
BEGIN DESCRIPTION:
Long Creek 70.0
END DESCRIPTION:
XS GIS Cut Line= 3
      1652991.29      6924512.16      1652505.00      6925488.00
      1652204.97      6925788.03
#Sta/Elev= 30
  3886.7 1745.89  3933.4 1741.97  4022.9 1738.88  4252.0 1736.51  4295.2 1735.89
  4425.8 1734.66  4463.0 1733.00  4476.2 1734.51  4627.3 1735.34  4789.5 1733.32
  4851.1 1733.31  4873.5 1732.85  4879.1 1731.92  4940.6 1731.32  4963.0 1730.21
  4974.2 1728.27  4975.6 1726.54  4976.1 1726.04  5006.7 1726.54  5012.4 1730.20
  5019.4 1731.49  5033.6 1735.62  5047.7 1736.86  5076.0 1737.94  5132.6 1738.52
  5175.0 1740.27  5203.3 1743.75  5245.7 1751.41  5274.0 1754.65  5401.3 1760.11
#Mann=5,-1,0
  3886.7    0.05       0  4252.0    0.12       0  4295.2    0.05       0
  4975.6    0.05       0  5006.7    0.05       0
Bank Sta=4975.6,5006.7
Exp/Cntr=0.3,0.1

Type RM Length L Ch R = 1,42871,526,526,526
BEGIN DESCRIPTION:
Long Creek 69.0
END DESCRIPTION:
XS GIS Cut Line= 3
      1652455.01      6924337.97      1652305.00      6924988.00
      1652105.01      6925737.98
#Sta/Elev= 30
  4359.2 1764.66  4383.2 1761.94  4390.0 1759.74  4410.5 1756.68  4461.9 1753.23
  4516.6 1747.59  4533.7 1743.37  4564.5 1739.48  4602.1 1737.34  4697.9 1734.87
  4923.7 1733.53  4933.9 1732.19  4944.2 1732.51  4975.0 1726.25  4985.3 1725.34
  4993.5 1722.58  4993.9 1722.08  5018.5 1722.58  5023.7 1727.23  5049.0 1729.62
  5089.1 1730.91  5140.2 1730.85  5164.1 1732.35  5212.6 1732.97  5434.5 1734.18
  5584.5 1737.78  5616.2 1741.23  5664.7 1752.37  5704.9 1755.69  5802.5 1760.19
#Mann=3,-1,0
  4359.2    0.05       0  4993.5    0.05       0  5018.5    0.05       0
Bank Sta=4993.5,5018.5
Exp/Cntr=0.3,0.1

Type RM Length L Ch R = 1,42345,495,495,495
BEGIN DESCRIPTION:
Long Creek 68.0
END DESCRIPTION:
XS GIS Cut Line= 3
      1651855.00      6924487.99      1651805.00      6924888.00
      1652004.99      6925687.95
#Sta/Elev= 30
  4597.7 1749.62  4640.5 1746.57  4668.3 1742.57  4688.4 1738.22  4728.7 1734.23
  4769.0 1732.56  4940.4 1730.85  4950.4 1729.25  4958.0 1725.90  4963.0 1725.47
  4970.6 1722.15  4982.7 1720.86  4983.2 1720.36  5013.9 1720.86  5018.9 1722.84
  5024.0 1722.20  5042.1 1729.50  5060.1 1731.38  5176.1 1730.77  5485.3 1733.10
  5588.4 1735.23  5619.3 1736.96  5629.6 1737.98  5637.3 1739.97  5642.5 1739.63
  5678.6 1748.37  5683.7 1748.31  5701.8 1750.94  5753.3 1754.71  5825.4 1758.50
#Mann=3,-1,0
  4597.7    0.05       0  4982.7    0.05       0  5013.9    0.05       0
Bank Sta=4982.7,5013.9
Exp/Cntr=0.3,0.1

Type RM Length L Ch R = 1,41850,602,602,602
BEGIN DESCRIPTION:
Long Creek 67.0
END DESCRIPTION:
XS GIS Cut Line= 3
      1651541.67      6924454.77      1651328.35      6924815.78
      1651255.00      6925538.04
#Sta/Elev= 30
  4558.7 1743.97  4639.3 1742.30  4660.7 1740.89  4713.4 1734.94  4777.8 1731.32
  4864.4 1730.43  4894.8 1727.73  4900.6 1729.62  4916.3 1730.47  4931.9 1726.85
  4945.8 1725.65  4959.2 1725.17  4969.0 1725.98  4974.7 1723.12  4975.2 1722.62
  5005.9 1723.12  5010.4 1725.26  5020.5 1725.75  5040.6 1729.51  5050.6 1730.45
  5121.0 1729.44  5181.3 1730.13  5472.8 1729.07  5533.1 1730.15  5556.9 1731.62
  5583.3 1740.84  5603.4 1743.89  5643.6 1746.99  5673.8 1747.60  5704.0 1750.31
#Mann=3,-1,0
  4558.7    0.05       0  4974.7    0.03       0  5005.9    0.05       0
Bank Sta=4974.7,5005.9
Exp/Cntr=0.3,0.1

Type RM Length L Ch R = 1,41248,594,594,594
BEGIN DESCRIPTION:
Long Creek 66.0
END DESCRIPTION:
XS GIS Cut Line= 3
      1650855.00      6924187.96      1650755.00      6924988.00
      1650755.00      6925538.04
#Sta/Elev= 30
  4200.5 1753.57  4238.3 1749.06  4261.0 1747.63  4422.2 1739.99  4502.9 1733.24
  4583.5 1729.58  4654.0 1728.07  4785.0 1728.94  4802.7 1727.08  4807.7 1728.60
  4845.5 1723.62  4883.3 1725.54  4926.1 1723.31  4963.9 1724.45  4986.6 1723.21
  4988.4 1722.11  4988.9 1721.61  5020.1 1722.11  5026.8 1725.08  5036.8 1726.47
  5076.8 1728.00  5226.8 1728.30  5266.8 1724.57  5306.8 1726.36  5336.8 1729.74
  5356.8 1736.96  5396.8 1742.79  5446.8 1746.42  5496.8 1747.73  5556.8 1751.73
#Mann=3,-1,0
  4200.5    0.05       0  4988.4    0.05       0  5020.1    0.05       0
Bank Sta=4988.4,5020.1
Exp/Cntr=0.3,0.1

Type RM Length L Ch R = 1,40654,567,567,567
BEGIN DESCRIPTION:
Long Creek 65.0
END DESCRIPTION:
XS GIS Cut Line= 3
      1650055.00      6924088.02      1650305.00      6925238.00
      1650505.02      6925588.04
#Sta/Elev= 30
  3801.5 1763.94  3852.7 1762.54  3903.8 1759.13  3944.8 1753.66  4012.3 1747.78
  4105.4 1736.06  4180.1 1729.62  4497.4 1724.82  4532.2 1719.96  4558.8 1723.54
  4630.4 1725.68  4753.2 1726.82  4916.9 1725.57  4968.1 1722.68  4981.2 1720.78
  4986.3 1716.53  4988.4 1716.37  4988.8 1715.87  5013.8 1716.37  5023.7 1721.60
  5029.5 1721.77  5045.3 1728.40  5051.0 1728.36  5066.9 1735.33  5072.6 1735.30
  5088.5 1739.12  5131.7 1740.96  5169.1 1744.60  5233.9 1745.65  5381.5 1752.38
#Mann=3,-1,0
  3801.5    0.05       0  4988.4    0.05       0  5013.8    0.05       0
Bank Sta=4988.4,5013.8
Exp/Cntr=0.3,0.1

Type RM Length L Ch R = 1,40087,584,584,584
BEGIN DESCRIPTION:
Long Creek 64.0
END DESCRIPTION:
XS GIS Cut Line= 3
      1649305.02      6924438.02      1649805.00      6925088.00
      1650055.03      6925438.04
#Sta/Elev= 30
  4180.6 1762.17  4223.2 1758.06  4281.2 1755.23  4395.1 1739.38  4422.5 1733.04
  4466.0 1727.84  4536.7 1725.17  4694.4 1723.56  4758.7 1717.71  4786.2 1718.73
  4808.6 1723.32  4914.5 1724.48  4943.5 1723.18  4958.1 1718.83  4964.4 1719.83
  4972.6 1717.63  4978.9 1718.95  4982.0 1716.58  4982.4 1716.08  5007.4 1716.58
  5008.0 1719.67  5037.5 1721.33  5100.2 1720.74  5236.6 1723.09  5251.3 1725.32
  5266.1 1731.91  5280.8 1734.32  5352.1 1739.76  5381.6 1739.66  5430.8 1742.79
#Mann=3,-1,0
  4180.6    0.05       0  4982.0    0.05       0  5007.4    0.05       0
Bank Sta=4982,5007.4
Exp/Cntr=0.3,0.1

Type RM Length L Ch R = 1,39503,566,566,566
BEGIN DESCRIPTION:
Long Creek 63.0
END DESCRIPTION:
XS GIS Cut Line= 3
      1648955.00      6924788.00      1649305.00      6925288.00
      1649554.98      6925787.96
#Sta/Elev= 30
  4388.9 1756.80  4425.5 1752.75  4453.0 1747.31  4474.3 1745.91  4518.4 1739.82
  4554.1 1728.23  4619.5 1715.66  4640.4 1719.48  4697.1 1722.96  4711.9 1722.09
  4905.5 1722.45  4962.6 1720.93  4970.9 1717.32  4977.0 1716.66  4984.2 1712.16
  4984.6 1711.66  5009.7 1712.16  5021.6 1715.32  5030.0 1719.34  5035.6 1718.76
  5043.9 1722.03  5057.9 1722.28  5074.7 1720.47  5125.0 1723.03  5178.1 1721.32
  5200.5 1722.48  5236.8 1721.59  5334.6 1724.99  5401.7 1731.45  5558.2 1737.24
#Mann=3,-1,0
  4388.9    0.05       0  4984.2    0.05       0  5009.7    0.05       0
Bank Sta=4984.2,5009.7
Exp/Cntr=0.3,0.1

Type RM Length L Ch R = 1,38937,579,579,579
BEGIN DESCRIPTION:
Long Creek 62.0
END DESCRIPTION:
XS GIS Cut Line= 3
      1648655.00      6924988.00      1648805.00      6925488.00
      1649555.00      6926288.00
#Sta/Elev= 30
  4482.9 1754.07  4514.2 1751.20  4556.0 1745.44  4609.1 1741.18  4642.1 1737.04
  4670.0 1732.17  4681.3 1727.92  4708.2 1720.76  4741.3 1716.15  4754.3 1716.25
  4785.7 1720.09  4806.5 1720.99  4845.7 1719.84  4942.3 1721.10  4955.3 1720.09
  4963.2 1717.29  4973.6 1715.29  4977.9 1712.80  4978.3 1712.30  5003.4 1712.80
  5004.9 1714.17  5018.8 1716.62  5075.5 1720.09  5118.0 1720.09  5160.5 1718.05
  5273.8 1722.80  5422.3 1726.07  5669.9 1734.56  5981.1 1748.21  6101.5 1756.61
#Mann=3,-1,0
  4482.9    0.05       0  4977.9    0.03       0  5003.4    0.05       0
Bank Sta=4977.9,5003.4
Exp/Cntr=0.3,0.1

Type RM Length L Ch R = 1,38358,586,586,586
BEGIN DESCRIPTION:
Long Creek 61.0
END DESCRIPTION:
XS GIS Cut Line= 3
      1648355.00      6925088.03      1648405.00      6925838.00
      1649204.97      6926437.98
#Sta/Elev= 30
  4248.0 1751.93  4278.0 1750.43  4378.3 1740.92  4428.4 1738.54  4488.5 1732.19
  4538.6 1728.85  4628.8 1717.75  4658.9 1715.79  4678.9 1715.01  4699.0 1717.93
  4759.1 1715.10  4769.1 1716.73  4799.2 1717.82  4889.4 1717.60  4969.6 1714.64
  4993.6 1710.70  4994.0 1710.20  5016.0 1710.70  5042.3 1716.40  5056.9 1715.19
  5063.2 1716.98  5086.1 1715.89  5149.6 1718.29  5177.8 1720.72  5277.8 1721.77
  5527.8 1728.86  5649.6 1734.93  5713.2 1735.93  5821.5 1740.80  5999.6 1752.22
#Mann=3,-1,0
  4248.0    0.05       0  4993.6    0.03       0  5016.0    0.05       0
Bank Sta=4993.6,5016
Exp/Cntr=0.3,0.1

Type RM Length L Ch R = 1,37772,546,546,546
BEGIN DESCRIPTION:
Long Creek 60.0
END DESCRIPTION:
XS GIS Cut Line= 3
      1648104.99      6925138.04      1648005.00      6925588.00
      1647605.00      6926687.99
#Sta/Elev= 30
  4539.9 1746.71  4607.7 1740.14  4656.4 1738.40  4699.9 1734.70  4714.0 1734.88
  4765.2 1729.79  4840.8 1726.72  4933.0 1717.95  4970.1 1710.97  4995.8 1710.53
  4996.2 1710.03  5021.6 1710.53  5032.8 1714.29  5041.4 1715.52  5064.7 1713.56
  5072.0 1714.83  5127.9 1716.52  5189.0 1716.99  5320.1 1714.87  5397.9 1716.47
  5469.0 1716.11  5522.2 1714.28  5540.2 1716.69  5749.0 1719.02  5835.5 1724.11
  5921.9 1734.77  5983.1 1739.46  6039.0 1746.49  6107.5 1750.99  6171.3 1752.63
#Mann=3,-1,0
  4539.9    0.05       0  4995.8    0.03       0  5021.6    0.05       0
Bank Sta=4995.8,5021.6
Exp/Cntr=0.3,0.1

Type RM Length L Ch R = 1,37226,663,663,663
BEGIN DESCRIPTION:
Long Creek 59.0
END DESCRIPTION:
XS GIS Cut Line= 3
      1647505.00      6924988.01      1647505.00      6925438.00
      1647555.00      6926688.01
#Sta/Elev= 30
  4544.3 1744.27  4664.3 1735.32  4804.3 1727.66  4894.3 1724.11  4944.3 1718.49
  4991.8 1709.64  5014.3 1710.12  5014.5 1708.78  5015.0 1708.28  5040.4 1708.78
  5044.3 1710.39  5074.4 1711.90  5104.4 1711.65  5154.4 1714.35  5204.5 1713.28
  5244.5 1714.61  5274.5 1713.63  5314.5 1714.75  5424.6 1713.26  5514.7 1714.25
  5564.7 1712.37  5614.8 1714.94  5774.9 1716.81  5814.9 1718.18  5845.0 1719.71
  5935.0 1731.11  6015.1 1738.22  6095.2 1747.15  6165.2 1751.04  6245.3 1752.89
#Mann=3,-1,0
  4544.3    0.05       0  5014.5    0.03       0  5040.4    0.05       0
Bank Sta=5014.5,5040.4
Exp/Cntr=0.3,0.1

Type RM Length L Ch R = 1,36563,425,425,425
BEGIN DESCRIPTION:
Long Creek 58.0
END DESCRIPTION:
XS GIS Cut Line= 3
      1646955.00      6924938.01      1646963.16      6925732.03
      1647438.11      6926384.39
#Sta/Elev= 30
  4125.6 1742.94  4355.6 1725.83  4405.6 1720.57  4435.6 1715.06  4485.6 1707.93
  4575.6 1712.23  4715.6 1712.67  4755.6 1712.30  4765.6 1711.28  4795.6 1712.17
  4885.6 1710.26  4932.3 1710.32  4976.3 1706.95  4977.9 1705.35  4978.4 1704.85
  5004.2 1705.35  5018.0 1707.06  5032.7 1710.28  5062.1 1712.48  5168.7 1711.28
  5204.2 1712.62  5375.8 1714.09  5511.8 1717.39  5562.0 1719.49  5591.4 1723.17
  5597.5 1722.54  5606.0 1723.97  5662.4 1726.85  5677.1 1729.57  5726.6 1733.67
#Mann=3,-1,0
  4125.6    0.05       0  4977.9    0.03       0  5004.2    0.05       0
Bank Sta=4977.9,5004.2
Exp/Cntr=0.3,0.1

Type RM Length L Ch R = 1,36138,603,603,603
BEGIN DESCRIPTION:
Long Creek 57.0
END DESCRIPTION:
XS GIS Cut Line= 3
      1646705.01      6925037.96      1646605.00      6925838.00
      1646505.01      6926437.96
#Sta/Elev= 30
  4205.2 1735.72  4243.0 1731.24  4295.9 1727.57  4328.7 1723.94  4396.7 1712.47
  4457.2 1710.04  4484.9 1706.81  4507.6 1709.83  4527.7 1710.49  4588.2 1710.80
  4651.2 1709.43  4668.8 1710.44  4749.4 1709.59  4930.8 1710.40  4951.0 1708.39
  4961.1 1704.82  4981.2 1704.62  4987.9 1702.57  4988.3 1702.07  5014.3 1702.57
  5039.3 1708.93  5044.4 1708.23  5082.4 1711.38  5173.7 1712.73  5287.7 1716.80
  5335.9 1721.10  5409.4 1724.12  5447.4 1728.09  5569.1 1736.61  5619.7 1741.32
#Mann=3,-1,0
  4205.2    0.05       0  4987.9    0.05       0  5014.3    0.05       0
Bank Sta=4987.9,5014.3
Exp/Cntr=0.3,0.1

Type RM Length L Ch R = 1,35535,564,564,564
BEGIN DESCRIPTION:
Long Creek 56.0
END DESCRIPTION:
XS GIS Cut Line= 3
      1646555.00      6924938.00      1646055.00      6925738.00
      1645854.98      6926338.05
#Sta/Elev= 30
  4043.3 1740.24  4224.3 1725.99  4276.2 1719.38  4318.7 1716.06  4349.3 1709.99
  4361.7 1709.22  4580.4 1707.26  4617.0 1708.13  4680.7 1706.56  4703.7 1708.10
  4732.6 1706.89  4769.1 1707.98  4833.4 1706.93  4878.8 1703.88  4915.4 1706.27
  4927.7 1708.68  4942.5 1708.01  4957.8 1704.43  4979.0 1703.18  4983.7 1700.36
  4993.0 1698.79  4993.4 1698.29  5019.4 1698.79  5028.9 1704.19  5071.0 1708.16
  5239.7 1710.48  5345.1 1715.30  5440.0 1722.98  5577.0 1737.39  5619.2 1740.03
#Mann=3,-1,0
  4043.3    0.05       0  4993.0    0.03       0  5019.4    0.05       0
Bank Sta=4993,5019.4
Exp/Cntr=0.3,0.1

Type RM Length L Ch R = 1,34971,317,317,317
BEGIN DESCRIPTION:
Long Creek 55.0
END DESCRIPTION:
XS GIS Cut Line= 3
      1646304.99      6924888.01      1645505.00      6925688.00
      1645354.99      6926088.04
#Sta/Elev= 30
  3868.1 1734.56  3924.7 1730.53  3952.9 1727.63  4051.9 1721.44  4094.4 1718.03
  4165.1 1714.70  4306.5 1700.53  4320.6 1700.28  4405.5 1706.99  4433.8 1707.03
  4462.1 1706.97  4490.3 1705.52  4674.2 1706.44  4900.5 1705.61  4928.7 1703.67
  4957.0 1703.08  4971.2 1701.09  5029.0 1699.76  5029.5 1699.26  5055.5 1699.76
  5063.5 1699.83  5094.7 1706.21  5100.0 1705.31  5106.3 1706.52  5180.1 1709.65
  5255.8 1715.91  5309.2 1723.26  5341.2 1726.31  5394.6 1733.38  5426.7 1735.86
#Mann=3,-1,0
  3868.1    0.05       0  5029.0    0.03       0  5055.5    0.05       0
Bank Sta=5029,5055.5
Exp/Cntr=0.3,0.1

Type RM Length L Ch R = 1,34654,374,374,374
BEGIN DESCRIPTION:
Long Creek 54.0
END DESCRIPTION:
XS GIS Cut Line= 3
      1645929.31      6924599.70      1645242.80      6925540.57
      1645116.99      6925890.65
#Sta/Elev= 30
  3838.4 1722.44  3954.9 1718.84  3990.5 1716.51  4120.2 1713.29  4206.0 1707.24
  4262.4 1699.30  4297.9 1698.99  4319.1 1704.37  4348.1 1705.67  4548.9 1705.10
  4591.4 1703.54  4670.2 1703.73  4720.4 1702.57  4735.1 1700.90  4756.0 1702.42
  4806.2 1701.67  4835.5 1703.37  4877.2 1701.59  4927.4 1701.64  4950.4 1703.03
  4997.8 1696.37  4998.3 1695.87  5024.3 1696.37  5053.5 1703.50  5156.8 1704.51
  5249.0 1709.55  5279.7 1713.10  5310.5 1719.20  5361.3 1724.67  5375.1 1727.37
#Mann=3,-1,0
  3838.4    0.05       0  4997.8    0.03       0  5024.3    0.05       0
Bank Sta=4997.8,5024.3
Exp/Cntr=0.3,0.1

Type RM Length L Ch R = 1,34280,298,298,298
BEGIN DESCRIPTION:
Mapping XS 1f174a55
END DESCRIPTION:
XS GIS Cut Line= 3
      1645103.09      6924034.67      1644919.06      6925395.80
      1644842.67      6925829.81
#Sta/Elev= 30
  3614.9 1722.12  3786.0 1716.59  4102.6 1710.21  4445.7 1706.28  4506.3 1698.41
  4532.5 1696.74  4537.6 1699.19  4546.6 1699.86  4597.1 1699.87  4617.3 1702.17
  4687.9 1702.01  4798.9 1700.18  4839.3 1697.29  4879.6 1697.41  4889.7 1694.67
  4899.8 1694.40  4930.1 1699.58  4960.4 1701.10  4983.5 1698.20  4987.4 1693.78
  4987.9 1693.28  5013.9 1693.78  5021.1 1697.64  5038.5 1700.05  5112.5 1700.04
  5183.6 1704.81  5275.7 1718.64  5295.3 1719.90  5366.3 1729.24  5429.1 1732.69
#Mann=3,-1,0
  3614.9    0.05       0  4987.4    0.03       0  5013.9    0.05       0
Bank Sta=4987.4,5013.9
Exp/Cntr=0.3,0.1

Type RM Length L Ch R = 1,33982,515,515,515
BEGIN DESCRIPTION:
Long Creek 53.0
END DESCRIPTION:
XS GIS Cut Line= 3
      1644544.06      6923968.74      1644620.45      6925392.33
      1644705.01      6925688.04
#Sta/Elev= 30
  3585.7 1723.58  3705.1 1715.70  3775.2 1713.56  4065.2 1708.50  4306.0 1707.56
  4456.2 1701.75  4630.6 1700.29  4676.5 1701.48  4796.7 1698.68  4826.7 1699.27
  4876.8 1697.59  4896.8 1694.46  4916.9 1694.68  4926.9 1693.22  4956.9 1695.37
  4977.0 1695.26  4984.3 1693.00  4984.8 1692.50  5010.8 1693.00  5011.3 1695.14
  5017.2 1698.44  5078.4 1703.34  5083.6 1702.61  5142.0 1707.88  5204.5 1711.35
  5224.0 1714.79  5229.2 1714.40  5263.0 1719.20  5287.7 1720.87  5318.9 1724.89
#Mann=3,-1,0
  3585.7    0.05       0  4984.3    0.05       0  5010.8    0.05       0
Bank Sta=4984.3,5010.8
Exp/Cntr=0.3,0.1

Type RM Length L Ch R = 1,33467,197,197,197
BEGIN DESCRIPTION:
Mapping XS 301bb2bd
END DESCRIPTION:
XS GIS Cut Line= 3
      1644033.64      6924211.77      1644137.81      6925388.85
      1644570.91      6925828.88
#Sta/Elev= 30
  3919.3 1724.25  3975.8 1721.39  4025.9 1717.55  4096.2 1713.99  4108.1 1712.60
  4166.5 1710.73  4206.6 1710.41  4226.7 1709.26  4708.6 1697.83  4859.2 1697.06
  4896.7 1695.09  4919.4 1696.26  4949.5 1696.73  4959.6 1696.30  4969.6 1693.36
  4973.0 1689.03  4973.6 1688.53  5005.7 1688.53  5006.3 1689.03  5008.6 1689.92
  5013.6 1689.33  5019.8 1691.32  5029.9 1692.84  5155.0 1698.62  5190.3 1701.82
  5296.3 1705.21  5352.9 1708.56  5565.1 1716.36  5664.1 1722.98  5718.4 1725.86
#Mann=3,-1,0
  3919.3    0.05       0  4973.0    0.05       0  5006.3    0.05       0
Bank Sta=4973,5006.3
Exp/Cntr=0.3,0.1

Type RM Length L Ch R = 1,33270,564,564,564
BEGIN DESCRIPTION:
Mapping XS 91bb8bac
END DESCRIPTION:
XS GIS Cut Line= 4
      1643760.94      6924869.34      1643809.67      6925129.24
      1643919.33      6925267.33      1644073.67      6925657.23
#Sta/Elev= 30
  4483.8 1699.38  4530.6 1697.66  4535.7 1697.94  4543.5 1697.51  4604.5 1696.60
  4765.3 1696.13  4887.1 1695.10  4928.5 1695.26  4936.0 1694.10  4941.5 1690.64
  4942.1 1690.14  4974.3 1690.14  4974.9 1690.64  4982.6 1691.04  5000.6 1690.83
  5022.1 1692.84  5031.3 1694.06  5036.6 1694.19  5043.6 1695.13  5066.4 1695.91
  5090.7 1696.11  5108.1 1696.98  5115.0 1697.76  5139.4 1698.81  5228.5 1701.36
  5247.5 1701.57  5252.9 1701.97  5306.9 1702.88  5323.2 1702.81  5343.9 1703.47
#Mann=3,-1,0
  4483.8    0.05       0  4941.5    0.03       0  4974.9    0.05       0
Bank Sta=4941.5,4974.9
Exp/Cntr=0.3,0.1

Type RM Length L Ch R = 1,32706,338,338,338
BEGIN DESCRIPTION:
Long Creek 52.0
END DESCRIPTION:
XS GIS Cut Line= 3
      1643205.01      6925038.01      1643405.00      6925388.00
      1644804.97      6926037.99
#Sta/Elev= 30
  4606.8 1730.01  4673.7 1729.43  4679.5 1727.12  4775.9 1725.20  4781.7 1721.64
  4797.5 1719.75  4803.3 1716.56  4813.4 1715.76  4819.1 1712.86  4878.2 1705.35
  4894.0 1701.88  4899.8 1697.74  4921.4 1689.06  4937.2 1688.10  4943.0 1690.19
  4958.8 1687.68  4986.9 1687.60  4990.3 1685.43  4990.9 1684.93  5023.8 1685.43
  5047.0 1688.43  5069.9 1687.28  5098.3 1690.31  5189.9 1693.34  5424.4 1696.39
  5891.9 1707.10  6116.0 1715.66  6213.1 1723.02  6396.3 1732.44  6553.4 1735.22
#Mann=3,-1,0
  4606.8    0.05       0  4990.3    0.03       0  5023.8    0.05       0
Bank Sta=4990.3,5023.8
Exp/Cntr=0.3,0.1

Type RM Length L Ch R = 1,32368,175,175,175
BEGIN DESCRIPTION:
Mapping XS 77403b84
END DESCRIPTION:
XS GIS Cut Line= 3
      1643050.99      6925527.73      1643214.20      6925645.80
      1644287.12      6925972.19
#Sta/Elev= 30
  4804.5 1715.96  4858.7 1715.28  4900.4 1711.34  4929.8 1707.19  4950.7 1705.86
  4965.4 1700.71  4971.6 1700.67  4980.1 1692.14  4986.3 1690.34  4990.5 1681.11
  4990.9 1680.61  5010.6 1681.11  5031.8 1683.46  5038.1 1687.83  5048.6 1690.75
  5079.9 1688.55  5174.0 1693.09  5206.5 1693.08  5226.3 1694.93  5234.2 1692.58
  5239.4 1693.61  5247.2 1692.75  5267.0 1693.94  5487.6 1695.87  5602.6 1699.41
  5863.9 1702.21  5960.8 1704.35  6041.6 1707.63  6083.4 1707.89  6127.4 1710.21
#Mann=3,-1,0
  4804.5    0.05       0  4990.5    0.03       0  5010.6    0.05       0
Bank Sta=4990.5,5010.6
Exp/Cntr=0.3,0.1

Type RM Length L Ch R = 1,32193,144,144,144
BEGIN DESCRIPTION:
Mapping XS 0b9533dd
END DESCRIPTION:
XS GIS Cut Line= 3
      1643039.46      6925718.12      1643173.26      6925809.67
      1643870.19      6925961.02
#Sta/Elev= 30
  4804.9 1707.38  4815.6 1706.60  4866.4 1705.85  4908.5 1703.13  4932.1 1700.59
  4938.2 1700.89  4944.9 1696.81  4953.1 1687.51  4959.1 1687.28  4965.1 1678.49
  4966.7 1673.90  4967.3 1673.40  4999.5 1673.40  5000.2 1673.90  5009.7 1681.47
  5027.5 1688.39  5032.6 1688.08  5076.6 1697.51  5120.6 1700.05  5132.5 1699.53
  5153.0 1693.69  5163.2 1692.52  5234.9 1693.48  5296.3 1692.97  5306.5 1693.67
  5312.1 1695.23  5317.2 1694.16  5347.4 1693.26  5449.3 1696.44  5680.2 1699.09
#Mann=3,-1,0
  4804.9    0.05       0  4966.7    0.03       0  5000.2    0.05       0
Bank Sta=4966.7,5000.2
Exp/Cntr=0.3,0.1

Type RM Length L Ch R = 1,32049,389,389,389
BEGIN DESCRIPTION:
Mapping XS 47455cc2
END DESCRIPTION:
XS GIS Cut Line= 3
      1643005.89      6925760.41      1643193.36      6925958.30
      1644051.32      6926118.60
#Sta/Elev= 30
  4715.1 1705.54  4854.2 1702.77  4903.9 1699.84  4910.8 1697.65  4918.1 1697.96
  4925.0 1690.50  4939.1 1690.12  4946.0 1680.94  4953.3 1681.94  4957.6 1673.89
  4958.2 1673.39  4991.1 1673.89  5009.0 1678.13  5014.0 1678.17  5019.9 1681.26
  5050.4 1690.24  5101.3 1696.02  5152.1 1692.36  5287.5 1692.12  5392.8 1694.35
  5457.3 1693.80  5503.2 1695.23  5508.3 1694.60  5538.7 1695.42  5608.5 1695.49
  5613.6 1694.68  5762.5 1697.76  5776.7 1696.92  5829.3 1698.29  5860.5 1698.18
#Mann=3,-1,0
  4715.1    0.05       0  4957.6    0.03       0  4991.1    0.05       0
Bank Sta=4957.6,4991.1
Exp/Cntr=0.3,0.1

Type RM Length L Ch R = 1,31660,283,283,283
BEGIN DESCRIPTION:
Mapping XS 76eab61b
END DESCRIPTION:
XS GIS Cut Line= 3
      1642991.97      6925996.48      1643020.37      6926259.18
      1643726.67      6926703.94
#Sta/Elev= 30
  4617.4 1696.22  4830.2 1693.97  4890.9 1692.24  4898.9 1693.04  4942.7 1689.07
  4985.1 1687.14  5006.3 1684.68  5015.7 1685.24  5021.6 1684.42  5036.9 1685.88
  5058.1 1686.74  5094.6 1685.38  5100.5 1685.77  5115.8 1684.55  5120.2 1683.02
  5120.8 1682.52  5153.1 1682.52  5153.7 1683.02  5158.9 1685.77  5167.6 1686.39
  5173.5 1689.75  5377.1 1689.74  5456.0 1690.69  5501.6 1692.18  5523.1 1695.15
  5550.2 1701.15  5586.7 1707.80  5596.1 1708.70  5602.0 1710.41  5716.3 1718.01
#Mann=3,-1,0
  4617.4    0.05       0  5120.2    0.05       0  5153.7    0.05       0
Bank Sta=5120.2,5153.7
Exp/Cntr=0.3,0.1

Type RM Length L Ch R = 1,31377,210,210,210
BEGIN DESCRIPTION:
Mapping XS 695ce580
END DESCRIPTION:
XS GIS Cut Line= 3
      1642964.18      6926065.98      1642856.56      6926430.52
      1643255.17      6926953.92
#Sta/Elev= 30
  4489.6 1694.99  4754.6 1692.49  4959.3 1688.78  4967.1 1688.46  4980.2 1684.59
  4994.7 1682.88  5030.1 1686.14  5056.9 1680.27  5057.5 1679.77  5090.4 1680.27
  5094.5 1682.10  5117.3 1686.02  5138.1 1687.80  5194.3 1685.41  5244.2 1687.61
  5294.1 1687.45  5323.2 1689.54  5331.4 1693.53  5337.7 1694.10  5344.2 1699.75
  5352.2 1703.68  5358.5 1703.08  5381.3 1707.77  5387.6 1707.78  5402.1 1713.70
  5408.4 1713.45  5416.7 1716.60  5423.0 1716.81  5431.2 1719.32  5527.6 1722.88
#Mann=3,-1,0
  4489.6    0.05       0  5056.9    0.05       0  5090.4    0.05       0
Bank Sta=5056.9,5090.4
Exp/Cntr=0.3,0.1

Type RM Length L Ch R = 1,31167,340,340,340
BEGIN DESCRIPTION:
Long Creek 51.0
END DESCRIPTION:
XS GIS Cut Line= 3
      1642821.16      6926032.58      1642703.97      6926550.84
      1643055.00      6926988.00
#Sta/Elev= 30
  4264.1 1694.14  4363.6 1692.21  4556.7 1691.40  4676.0 1688.84  4761.8 1688.51
  4767.5 1687.80  4900.9 1685.83  4936.1 1686.01  4958.5 1684.66  4964.9 1683.32
  4971.4 1680.01  4986.5 1678.73  4987.0 1678.23  5013.6 1678.73  5014.5 1679.54
  5028.9 1680.86  5049.7 1684.93  5086.5 1683.64  5099.6 1684.76  5107.3 1689.38
  5113.7 1688.40  5121.7 1694.39  5128.1 1695.42  5136.1 1698.81  5150.5 1700.06
  5171.3 1703.68  5264.1 1709.61  5299.3 1712.67  5305.7 1714.13  5356.1 1715.38
#Mann=3,-1,0
  4264.1    0.05       0  4986.5    0.05       0  5013.6    0.05       0
Bank Sta=4986.5,5013.6
Exp/Cntr=0.3,0.1

Type RM Length L Ch R = 1,30827,368,368,368
BEGIN DESCRIPTION:
Mapping XS f84d5abc
END DESCRIPTION:
XS GIS Cut Line= 3
      1642839.20      6925895.79      1642551.00      6926697.88
      1642395.20      6927234.52
#Sta/Elev= 30
  4152.8 1696.47  4399.5 1691.62  4564.4 1691.09  4760.8 1687.59  4922.4 1685.59
  4941.5 1684.43  4962.7 1681.14  4973.3 1681.84  4984.0 1677.44  4993.9 1675.07
  4994.5 1674.57  5020.8 1674.57  5021.4 1675.07  5026.0 1678.29  5043.1 1680.34
  5048.3 1680.01  5057.3 1680.79  5076.7 1689.17  5081.9 1688.84  5088.5 1690.91
  5098.9 1691.44  5115.4 1694.33  5182.2 1696.50  5221.3 1699.99  5259.8 1702.07
  5307.2 1707.67  5332.4 1708.47  5390.5 1712.13  5510.5 1716.13  5563.9 1717.15
#Mann=3,-1,0
  4152.8    0.05       0  4993.9    0.03       0  5021.4    0.05       0
Bank Sta=4993.9,5021.4
Exp/Cntr=0.3,0.1

Type RM Length L Ch R = 1,30459,289,289,289
BEGIN DESCRIPTION:
Long Creek 50.0
END DESCRIPTION:
XS GIS Cut Line= 3
      1642854.99      6925688.01      1642255.00      6926488.00
      1642055.00      6926838.00
#Sta/Elev= 30
  3973.9 1705.20  4052.0 1702.56  4160.3 1695.97  4202.0 1694.63  4381.2 1691.05
  4523.9 1689.08  4537.4 1689.97  4566.6 1688.47  4652.0 1686.99  4773.9 1686.18
  4895.8 1683.86  4923.9 1681.70  4960.3 1681.85  4966.6 1678.16  4967.5 1674.28
  4968.0 1673.78  4991.5 1674.28  4996.9 1676.95  5009.2 1675.60  5031.5 1674.67
  5046.6 1676.35  5054.5 1676.29  5062.4 1679.44  5068.2 1683.63  5089.8 1695.51
  5121.5 1702.10  5135.1 1706.98  5148.8 1710.30  5238.8 1713.97  5377.0 1716.27
#Mann=3,-1,0
  3973.9    0.05       0  4967.5    0.05       0  4991.5    0.05       0
Bank Sta=4967.5,4991.5
Exp/Cntr=0.3,0.1

Type RM Length L Ch R = 1,30170,319,319,319
BEGIN DESCRIPTION:
Mapping XS d13180ce
END DESCRIPTION:
XS GIS Cut Line= 3
      1642547.50      6925829.85      1642037.30      6926308.66
      1641735.00      6926572.91
#Sta/Elev= 30
  4292.6 1693.43  4547.7 1687.95  4795.3 1684.73  4873.0 1682.97  4915.5 1681.51
  4972.1 1676.83  4979.4 1674.94  4986.3 1672.18  4986.6 1669.81  4987.2 1669.31
  5014.1 1669.81  5014.7 1671.85  5049.8 1676.74  5057.4 1679.81  5071.6 1688.29
  5078.3 1690.30  5100.1 1693.98  5106.7 1696.28  5149.5 1698.16  5156.1 1699.45
  5170.3 1700.35  5177.9 1699.91  5213.0 1701.70  5241.5 1701.80  5319.4 1704.08
  5347.8 1703.53  5354.5 1704.36  5362.1 1703.67  5382.9 1704.63  5393.8 1704.06
#Mann=3,-1,0
  4292.6    0.05       0  4986.6    0.05       0  5014.1    0.05       0
Bank Sta=4986.6,5014.1
Exp/Cntr=0.3,0.1

Type RM Length L Ch R = 1,29851,483,483,483
BEGIN DESCRIPTION:
Mapping XS a1b6ccd7
END DESCRIPTION:
XS GIS Cut Line= 4
      1642217.59      6925900.93      1641987.82      6926076.89
      1641628.45      6926066.47      1641234.76      6926307.04
#Sta/Elev= 30
  4547.8 1686.67  4835.8 1681.97  4870.0 1684.92  4900.1 1684.90  4920.1 1680.16
  4940.1 1679.24  4950.1 1677.16  4968.2 1667.33  4973.2 1670.65  4978.3 1666.54
  4978.9 1666.04  5005.8 1666.54  5030.1 1670.08  5050.1 1675.13  5090.1 1680.68
  5110.1 1681.91  5170.2 1682.80  5207.9 1682.00  5213.8 1682.77  5266.0 1682.75
  5287.3 1683.99  5302.8 1682.38  5345.4 1683.84  5360.8 1683.07  5470.3 1686.18
  5492.4 1688.74  5550.5 1691.38  5599.2 1692.18  5645.3 1694.20  5658.1 1693.79
#Mann=3,-1,0
  4547.8    0.05       0  4978.3    0.05       0  5005.8    0.05       0
Bank Sta=4978.3,5005.8
Exp/Cntr=0.3,0.1

Type RM Length L Ch R = 1,29368,656,656,656
BEGIN DESCRIPTION:
Long Creek 48.0
END DESCRIPTION:
XS GIS Cut Line= 3
      1641990.44      6925399.79      1641805.00      6925638.00
      1641165.50      6926193.56
#Sta/Elev= 30
  4718.3 1705.00  4735.2 1702.61  4764.1 1700.16  4770.5 1700.79  4799.4 1697.31
  4855.5 1694.38  4870.0 1692.92  4878.1 1690.87  4914.5 1687.45  4922.9 1686.61
  4948.7 1683.27  4977.7 1670.13  4984.0 1668.88  4984.9 1666.77  4985.5 1666.27
  5012.6 1666.77  5012.9 1670.43  5017.0 1673.45  5055.8 1677.29  5093.3 1678.43
  5094.8 1678.43  5176.4 1679.78  5227.7 1679.25  5235.5 1678.97  5324.9 1677.59
  5374.9 1678.40  5487.8 1682.78  5800.3 1689.27  5849.6 1691.01  5867.3 1692.99
#Mann=9,-1,0
  4718.3    0.05       0  4914.5    0.12       0  4922.9    0.05       0
  4984.9    0.05       0  5012.6    0.05       0  5093.3    0.12       0
  5094.8    0.05       0  5227.7    0.12       0  5235.5    0.05       0
Bank Sta=4984.9,5012.6
Exp/Cntr=0.3,0.1

Type RM Length L Ch R = 1,28712,559,559,559
BEGIN DESCRIPTION:
Mapping XS d024ac69
END DESCRIPTION:
XS GIS Cut Line= 3
      1641228.08      6925222.21      1641217.67      6925440.94
      1641141.28      6926159.71
#Sta/Elev= 30
  4758.6 1693.96  4764.4 1694.38  4774.4 1693.87  4804.4 1693.60  4814.5 1692.87
  4824.5 1692.93  4884.5 1691.21  4914.6 1689.08  4929.1 1684.28  4934.6 1677.85
  4954.6 1674.95  4964.6 1672.42  4973.6 1667.53  4977.6 1667.53  4981.9 1661.20
  4982.5 1660.70  5009.0 1660.70  5009.7 1661.20  5024.9 1666.89  5035.0 1673.04
  5045.0 1675.72  5055.1 1676.43  5111.8 1676.81  5155.6 1677.78  5185.8 1679.17
  5209.9 1679.17  5286.4 1680.88  5386.9 1682.27  5447.3 1683.67  5700.4 1690.65
#Mann=5,-1,0
  4758.6    0.05       0  4981.9    0.05       0  5009.7    0.05       0
  5111.8    0.12       0  5209.9    0.05       0
Bank Sta=4981.9,5009.7
Exp/Cntr=0.3,0.1

Type RM Length L Ch R = 1,28153,478,478,478
BEGIN DESCRIPTION:
Mapping XS 14997923
END DESCRIPTION:
XS GIS Cut Line= 3
      1641137.85      6925190.92      1640821.84      6925305.52
      1640444.07      6925693.68
#Sta/Elev= 30
  4445.9 1689.45  4570.3 1684.71  4595.6 1683.24  4619.1 1680.80  4743.4 1678.13
  4795.8 1675.24  4824.0 1672.25  4930.0 1670.06  4937.2 1669.13  4944.2 1669.43
  4951.4 1668.32  4958.3 1668.47  4976.5 1666.34  4977.2 1665.84  5011.2 1666.34
  5050.4 1667.01  5057.4 1668.58  5064.5 1673.92  5071.5 1673.34  5085.7 1675.83
  5128.1 1675.66  5149.2 1677.21  5163.4 1679.73  5170.5 1683.52  5198.8 1693.89
  5234.1 1702.15  5248.2 1704.76  5255.4 1705.04  5276.5 1707.88  5323.7 1709.60
#Mann=3,-1,0
  4445.9    0.05       0  4976.5    0.03       0  5011.2    0.05       0
Bank Sta=4976.5,5011.2
Exp/Cntr=0.3,0.1

Type RM Length L Ch R = 1,27675,263,263,263
BEGIN DESCRIPTION:
Long Creek 46.0
END DESCRIPTION:
XS GIS Cut Line= 3
      1641205.05      6925138.00      1640505.00      6925088.00
      1640380.00      6925163.00
#Sta/Elev= 30
  4318.5 1694.09  4328.6 1692.87  4408.8 1689.16  4438.9 1687.33  4458.9 1685.20
  4509.0 1682.84  4531.6 1682.77  4569.2 1681.07  4659.4 1679.05  4719.6 1678.59
  4849.9 1675.28  4930.1 1674.25  4960.2 1672.84  4980.2 1665.06  4986.3 1660.41
  4986.9 1659.91  5013.5 1659.91  5014.1 1660.41  5017.8 1665.01  5033.9 1665.44
  5055.3 1668.39  5065.0 1671.48  5070.9 1671.23  5086.4 1682.56  5092.2 1681.39
  5102.0 1687.51  5113.6 1692.05  5123.3 1694.43  5144.7 1696.47  5166.1 1696.66
#Mann=3,-1,0
  4318.5    0.05       0  4986.3    0.05       0  5014.1    0.05       0
Bank Sta=4986.3,5014.1
Exp/Cntr=0.3,0.1

Type RM Length L Ch R = 1,27412,329,329,329
BEGIN DESCRIPTION:
Mapping XS 376e874d
END DESCRIPTION:
XS GIS Cut Line= 2
      1641429.47      6924954.82      1640426.04      6924815.94
#Sta/Elev= 30
  4118.7 1701.18  4214.1 1698.35  4335.2 1692.99  4427.4 1688.00  4476.6 1683.97
  4547.2 1681.10  4566.0 1679.66  4577.5 1681.12  4587.6 1679.91  4607.8 1679.42
  4628.0 1680.24  4637.8 1679.78  4648.2 1678.06  4728.9 1677.22  4759.2 1675.64
  4819.8 1675.66  4951.0 1671.24  4961.1 1670.58  4971.2 1668.70  4981.3 1663.40
  4985.7 1658.39  4986.4 1657.89  5017.0 1658.39  5021.7 1659.60  5041.9 1668.20
  5062.1 1674.43  5078.7 1687.34  5083.8 1689.07  5092.4 1691.45  5131.7 1692.27
#Mann=3,-1,0
  4118.7    0.05       0  4985.7    0.03       0  5017.0    0.05       0
Bank Sta=4985.7,5017
Exp/Cntr=0.3,0.1

Type RM Length L Ch R = 1,27083,251,251,251
BEGIN DESCRIPTION:
Mapping XS a59000e5
END DESCRIPTION:
XS GIS Cut Line= 2
      1641266.28      6924673.58      1640464.22      6924479.14
#Sta/Elev= 30
  4306.3 1687.13  4310.8 1685.85  4338.5 1684.43  4352.6 1682.63  4410.5 1682.21
  4451.7 1680.31  4472.3 1681.19  4478.0 1680.17  4566.7 1677.83  4595.7 1678.21
  4636.9 1676.01  4708.9 1675.54  4832.4 1672.76  4853.0 1673.42  4906.3 1670.83
  4914.7 1669.59  4942.9 1669.22  4955.9 1667.30  4976.4 1660.43  4989.9 1659.27
  4990.9 1658.34  4991.6 1657.84  5022.2 1658.34  5026.5 1663.24  5031.7 1664.13
  5038.2 1669.02  5058.8 1678.25  5068.3 1680.71  5110.1 1684.31  5131.6 1684.96
#Mann=3,-1,0
  4306.3    0.05       0  4990.9    0.03       0  5022.2    0.05       0
Bank Sta=4990.9,5022.2
Exp/Cntr=0.3,0.1

Type RM Length L Ch R = 1,26832,469,469,469
BEGIN DESCRIPTION:
Mapping XS 2cbc1f7a
END DESCRIPTION:
XS GIS Cut Line= 2
      1641280.20      6924308.99      1640439.92      6924256.91
#Sta/Elev= 30
  4383.5 1697.13  4458.8 1690.65  4477.1 1686.74  4482.1 1687.06  4488.9 1684.39
  4498.9 1681.97  4529.0 1678.62  4539.0 1676.75  4579.1 1675.23  4619.2 1675.19
  4649.2 1674.13  4719.3 1673.34  4809.5 1673.25  4829.6 1672.03  4919.7 1670.77
  4949.8 1668.44  4959.8 1665.97  4965.1 1663.64  4970.1 1663.30  4972.5 1662.37
  4973.2 1661.87  5006.5 1661.87  5007.3 1662.37  5009.9 1663.50  5029.9 1665.72
  5040.0 1665.46  5080.0 1667.53  5126.0 1673.29  5190.2 1675.73  5225.4 1676.30
#Mann=3,-1,0
  4383.5    0.05       0  4972.5    0.03       0  5007.3    0.05       0
Bank Sta=4972.5,5007.3
Exp/Cntr=0.3,0.1

Type RM Length L Ch R = 1,26363,345,345,345
BEGIN DESCRIPTION:
Mapping XS 0a521c33
END DESCRIPTION:
XS GIS Cut Line= 4
      1641519.72      6923857.60      1640853.09      6923836.77
      1640714.20      6923861.08      1640429.71      6924214.94
#Sta/Elev= 30
  4313.3 1713.47  4438.1 1707.87  4461.9 1706.16  4508.1 1704.61  4588.2 1699.43
  4618.2 1699.23  4642.9 1697.10  4658.2 1695.11  4688.2 1692.82  4698.2 1689.98
  4728.2 1679.41  4748.2 1675.22  4777.0 1671.41  4828.3 1669.28  4923.3 1670.51
  4958.3 1669.65  4976.8 1665.57  4980.3 1665.57  4981.2 1661.12  4981.9 1660.62
  5015.3 1660.62  5016.1 1661.12  5125.8 1667.38  5175.4 1668.14  5282.6 1668.26
  5388.2 1669.90  5438.1 1671.48  5445.8 1671.05  5524.2 1674.53  5575.3 1675.34
#Mann=5,-1,0
  4313.3    0.05       0  4642.9    0.12       0  4923.3    0.05       0
  4981.2    0.03       0  5016.1    0.05       0
Bank Sta=4981.2,5016.1
Exp/Cntr=0.3,0.1

Type RM Length L Ch R = 1,26018,485,485,485
BEGIN DESCRIPTION:
Mapping XS 35447d89
END DESCRIPTION:
XS GIS Cut Line= 3
      1640693.36      6923253.43      1640735.03      6923732.60
      1640401.72      6924208.27
#Sta/Elev= 30
  4644.8 1710.87  4679.5 1707.41  4709.6 1701.85  4749.8 1684.96  4769.8 1679.30
  4789.9 1674.77  4836.0 1670.40  4910.4 1669.77  4930.4 1668.84  4940.5 1667.27
  4948.9 1664.80  4953.9 1665.18  4960.6 1663.14  4981.3 1660.38  4982.3 1659.88
  5019.1 1659.88  5020.1 1660.38  5020.8 1661.16  5030.8 1664.15  5040.9 1665.75
  5050.9 1666.34  5125.8 1666.40  5187.1 1664.49  5230.1 1667.11  5258.6 1667.91
  5359.7 1668.13  5466.9 1670.10  5510.9 1670.12  5603.8 1673.36  5706.6 1675.10
#Mann=3,-1,0
  4644.8    0.05       0  4981.3    0.03       0  5020.1    0.05       0
Bank Sta=4981.3,5020.1
Exp/Cntr=0.3,0.1

Type RM Length L Ch R = 1,25533,490,490,490
BEGIN DESCRIPTION:
Long Creek 45.0
END DESCRIPTION:
XS GIS Cut Line= 3
      1640055.02      6923288.03      1640255.00      6923638.00
      1640405.01      6924338.03
#Sta/Elev= 30
  4599.7 1718.83  4634.9 1717.77  4768.8 1709.59  4833.6 1702.68  4871.0 1697.10
  4892.6 1694.98  4899.1 1692.58  4914.2 1681.21  4930.1 1675.39  4935.8 1674.68
  4945.2 1670.77  4951.7 1666.32  4957.4 1664.98  4967.5 1660.47  4973.3 1659.13
  4975.8 1654.59  4976.6 1654.09  5006.0 1654.09  5006.8 1654.59  5027.5 1657.48
  5033.5 1661.96  5043.7 1665.53  5084.6 1668.74  5105.0 1669.39  5135.7 1668.61
  5370.9 1670.65  5493.7 1673.91  5600.2 1675.13  5649.6 1676.48  5718.7 1680.81
#Mann=3,-1,0
  4599.7    0.05       0  4975.8    0.05       0  5006.8    0.05       0
Bank Sta=4975.8,5006.8
Exp/Cntr=0.3,0.1

Type RM Length L Ch R = 1,25043,226,226,226
BEGIN DESCRIPTION:
Long Creek 44.0
END DESCRIPTION:
XS GIS Cut Line= 3
      1639805.00      6923437.99      1639805.00      6923838.00
      1640304.99      6924387.99
#Sta/Elev= 30
  4608.4 1713.37  4648.4 1710.98  4808.4 1697.03  4828.4 1696.24  4838.4 1695.23
  4848.4 1692.94  4888.4 1688.66  4898.4 1685.16  4908.4 1679.16  4918.4 1674.47
  4958.4 1657.89  4968.4 1654.48  4969.0 1653.45  4970.0 1652.95  5007.8 1653.45
  5022.3 1655.30  5036.5 1658.27  5043.9 1661.21  5050.6 1661.82  5064.8 1665.43
  5086.5 1667.40  5100.6 1667.75  5107.4 1666.70  5114.8 1667.12  5121.6 1666.37
  5355.4 1667.81  5489.9 1673.08  5581.8 1674.31  5695.3 1677.17  5751.7 1680.82
#Mann=3,-1,0
  4608.4    0.05       0  4969.0    0.05       0  5007.8    0.05       0
Bank Sta=4969,5007.8
Exp/Cntr=0.3,0.1

Type RM Length L Ch R = 1,24817,346,346,346
BEGIN DESCRIPTION:
Mapping XS ec379dd0
END DESCRIPTION:
XS GIS Cut Line= 4
      1639214.85      6923762.28      1639456.27      6923896.40
      1639779.85      6924005.38      1640297.88      6924442.94
#Sta/Elev= 30
  4513.7 1699.48  4598.6 1697.37  4642.1 1694.17  4674.0 1693.20  4717.6 1688.99
  4723.3 1686.29  4739.3 1683.76  4745.0 1681.41  4754.1 1680.52  4766.8 1677.28
  4782.8 1675.77  4786.4 1674.19  4838.9 1670.13  4883.5 1660.97  4933.4 1658.98
  4946.8 1660.16  4956.4 1658.23  4957.2 1657.73  4987.4 1658.23  4989.0 1659.86
  5010.1 1658.92  5020.7 1659.67  5041.8 1664.79  5064.7 1665.47  5371.4 1666.99
  5413.0 1668.46  5463.7 1672.02  5478.0 1671.53  5683.4 1675.84  5809.4 1681.58
#Mann=3,-1,0
  4513.7    0.05       0  4956.4    0.03       0  4987.4    0.05       0
Bank Sta=4956.4,4987.4
Exp/Cntr=0.3,0.1

Type RM Length L Ch R = 1,24471,281,281,281
BEGIN DESCRIPTION:
Long Creek 43.0
END DESCRIPTION:
XS GIS Cut Line= 3
      1639176.30      6923943.36      1639555.00      6924288.00
      1640355.02      6924688.01
#Sta/Elev= 30
  4479.7 1691.35  4517.7 1687.79  4531.9 1685.32  4545.6 1680.59  4588.0 1672.65
  4659.0 1665.62  4694.3 1664.62  4729.9 1660.72  4772.5 1663.93  4899.5 1662.29
  4927.9 1661.35  4935.3 1660.21  4942.1 1660.90  4963.7 1658.35  4994.5 1656.78
  4994.7 1655.71  4995.7 1655.21  5033.6 1655.71  5036.5 1657.79  5058.8 1662.47
  5072.8 1664.20  5318.8 1666.09  5341.1 1666.62  5380.3 1669.70  5654.2 1675.08
  5698.9 1676.89  5738.0 1680.08  5788.3 1681.53  5872.2 1687.93  5886.2 1688.13
#Mann=3,-1,0
  4479.7    0.05       0  4994.7    0.03       0  5033.6    0.05       0
Bank Sta=4994.7,5033.6
Exp/Cntr=0.3,0.1

Type RM Length L Ch R = 1,24190,272,272,272
BEGIN DESCRIPTION:
Mapping XS 757373df
END DESCRIPTION:
XS GIS Cut Line= 3
      1639158.64      6923982.61      1639443.36      6924527.74
      1640070.88      6925072.05
#Sta/Elev= 30
  4391.4 1689.09  4415.2 1687.48  4431.3 1684.40  4442.9 1679.84  4487.7 1672.34
  4547.7 1665.88  4630.3 1663.95  4829.1 1662.97  4917.4 1661.36  4927.7 1659.93
  4955.9 1652.90  4972.4 1652.33  4978.0 1653.96  4980.0 1651.19  4980.8 1650.69
  5011.1 1651.19  5014.8 1655.32  5021.8 1656.75  5035.7 1662.96  5049.9 1664.27
  5114.5 1664.36  5142.0 1663.35  5170.5 1664.21  5305.4 1664.18  5446.9 1665.39
  5780.2 1672.69  5787.9 1671.76  5794.5 1672.71  5802.1 1671.88  5837.1 1674.23
#Mann=3,-1,0
  4391.4    0.05       0  4980.0    0.03       0  5011.1    0.05       0
Bank Sta=4980,5011.1
Exp/Cntr=0.3,0.1

Type RM Length L Ch R = 1,23918,316,316,316
BEGIN DESCRIPTION:
Long Creek 42.0
END DESCRIPTION:
XS GIS Cut Line= 3
      1639054.99      6924237.96      1639205.00      6924638.00
      1639613.49      6925458.28
#Sta/Elev= 30
  4652.0 1681.93  4697.4 1676.16  4722.3 1674.71  4727.7 1672.38  4752.6 1669.25
  4790.9 1665.88  4807.8 1666.19  4813.1 1663.40  4868.3 1661.26  4953.7 1661.49
  4984.0 1656.72  4987.3 1653.81  4988.1 1653.31  5018.4 1653.81  5025.8 1657.29
  5087.6 1654.90  5110.0 1656.30  5132.4 1660.07  5160.4 1660.84  5624.9 1662.28
  5764.9 1664.86  5832.0 1671.65  5854.4 1676.22  5871.2 1682.05  5876.8 1682.22
  5883.6 1687.02  5893.6 1689.76  5921.6 1694.02  5928.3 1696.92  5995.6 1707.02
#Mann=3,-1,0
  4652.0    0.05       0  4987.3    0.03       0  5018.4    0.05       0
#XS Ineff=2,0
    0.00 4819.80 1672.73 5180.20    0.00 1672.73
Permanent Ineff=
       F       F
Bank Sta=4987.3,5018.4
Exp/Cntr=0.3,0.1

Type RM Length L Ch R = 1,23602,371,371,371
BEGIN DESCRIPTION:
Mapping XS 8feca8df
END DESCRIPTION:
XS GIS Cut Line= 3
      1638991.97      6924350.63      1638978.09      6924749.96
      1639213.62      6925404.61
#Sta/Elev= 30
  4529.8 1677.99  4584.4 1677.03  4807.3 1666.41  4948.5 1663.55  4959.2 1660.43
  4976.4 1652.36  4977.2 1651.86  5007.5 1652.36  5076.1 1654.03  5087.4 1656.90
  5107.5 1656.86  5129.2 1658.65  5138.2 1657.54  5174.2 1659.50  5255.7 1659.37
  5470.7 1661.57  5490.5 1664.03  5496.1 1665.72  5501.4 1665.34  5521.5 1670.07
  5526.8 1669.50  5552.2 1679.45  5557.5 1677.97  5564.9 1684.35  5582.9 1692.57
  5588.2 1692.15  5607.4 1697.07  5613.6 1699.95  5618.9 1699.55  5625.1 1701.94
#Mann=3,-1,0
  4529.8    0.05       0  4976.4    0.03       0  5007.5    0.05       0
#XS Ineff=2,0
    0.00 4830.00 1671.28 5170.00    0.00 1671.28
Permanent Ineff=
       F       F
Bank Sta=4976.4,5007.5
Exp/Cntr=0.3,0.1

Type RM Length L Ch R = 1,23231,498,498,498
BEGIN DESCRIPTION:
Long Creek 41.0
END DESCRIPTION:
XS GIS Cut Line= 3
      1638908.65      6924374.92      1638789.79      6925087.77
      1638703.77      6925371.53
#Sta/Elev= 30
  4270.4 1672.46  4321.1 1670.93  4326.1 1669.75  4344.5 1668.38  4386.9 1667.07
  4658.8 1661.14  4668.9 1661.56  4686.0 1660.38  4851.4 1658.18  4868.4 1656.20
  4881.8 1657.12  4922.4 1653.93  4952.8 1653.12  4983.2 1650.17  4987.4 1648.24
  4988.2 1647.74  5018.6 1648.24  5028.4 1650.92  5035.1 1654.44  5056.0 1658.70
  5066.5 1663.02  5087.4 1669.83  5094.2 1674.80  5099.4 1677.22  5108.3 1687.13
  5127.1 1694.24  5139.6 1697.40  5171.0 1702.56  5198.1 1704.38  5289.6 1703.35
#Mann=3,-1,0
  4270.4    0.05       0  4987.4    0.03       0  5018.6    0.05       0
Bank Sta=4987.4,5018.6
Exp/Cntr=0.3,0.1

Type RM Length L Ch R = 1,22733,584,584,584
BEGIN DESCRIPTION:
Long Creek 40.0
END DESCRIPTION:
XS GIS Cut Line= 3
      1638864.64      6924129.26      1638405.00      6924788.00
      1638329.16      6925004.45
#Sta/Elev= 30
  4196.5 1679.51  4223.8 1678.17  4259.5 1674.51  4316.9 1671.08  4366.8 1669.18
  4375.6 1667.68  4381.7 1667.98  4390.1 1666.96  4402.6 1666.82  4411.3 1667.69
  4804.8 1656.71  4849.3 1656.68  4855.4 1655.79  4950.5 1653.96  4971.4 1651.13
  4977.5 1648.80  4978.2 1645.79  4979.0 1645.29  5009.4 1645.79  5015.3 1646.86
  5020.9 1646.66  5046.3 1651.40  5063.3 1653.38  5084.5 1660.35  5108.3 1665.90
  5126.9 1671.35  5139.3 1676.89  5148.1 1679.86  5179.9 1683.91  5229.1 1683.79
#Mann=3,-1,0
  4196.5    0.05       0  4978.2    0.03       0  5009.4    0.05       0
Bank Sta=4978.2,5009.4
Exp/Cntr=0.3,0.1

Type RM Length L Ch R = 1,22149,564,564,564
BEGIN DESCRIPTION:
Long Creek 39.0
END DESCRIPTION:
XS GIS Cut Line= 3
      1638355.02      6923787.97      1638055.00      6924338.00
      1637855.01      6925087.96
#Sta/Elev= 30
  4373.2 1699.15  4453.0 1691.45  4534.1 1680.46  4578.3 1673.00  4703.6 1660.49
  4784.7 1654.99  4874.4 1653.64  4910.0 1648.97  4948.0 1650.93  4954.2 1649.71
  4955.5 1647.84  4956.3 1647.34  4987.0 1647.84  4991.7 1650.17  4996.9 1650.50
  5030.8 1650.00  5092.2 1652.55  5113.6 1651.77  5132.3 1647.97  5144.6 1648.42
  5212.5 1656.87  5227.4 1660.63  5268.8 1664.59  5299.9 1671.14  5327.7 1674.52
  5393.0 1672.13  5475.8 1673.49  5620.7 1682.36  5718.4 1685.91  5775.9 1690.36
#Mann=3,-1,0
  4373.2    0.05       0  4955.5    0.03       0  4987.0    0.05       0
Bank Sta=4955.5,4987
Exp/Cntr=0.3,0.1

Type RM Length L Ch R = 1,21585,562,562,562
BEGIN DESCRIPTION:
Long Creek 38.0
END DESCRIPTION:
XS GIS Cut Line= 3
      1637555.00      6923587.97      1637555.00      6924188.00
      1637754.98      6924587.96
#Sta/Elev= 30
  4422.3 1707.30  4472.3 1700.78  4542.3 1686.45  4562.3 1678.88  4572.3 1673.28
  4632.3 1660.58  4662.3 1657.45  4722.3 1648.22  4742.3 1647.73  4832.3 1651.53
  4932.3 1649.24  4952.3 1648.42  4982.3 1644.33  4983.6 1640.62  4984.2 1640.12
  5007.3 1640.62  5019.8 1644.44  5036.3 1645.26  5053.1 1652.43  5058.7 1651.75
  5067.1 1653.99  5170.5 1659.28  5187.2 1662.12  5192.8 1661.00  5209.6 1665.21
  5215.2 1664.36  5232.0 1667.95  5259.9 1668.00  5349.4 1673.96  5469.5 1671.84
#Mann=3,-1,0
  4422.3    0.05       0  4983.6    0.03       0  5007.3    0.05       0
Bank Sta=4983.6,5007.3
Exp/Cntr=0.3,0.1

Type RM Length L Ch R = 1,21023,575,575,575
BEGIN DESCRIPTION:
Long Creek 37.0
END DESCRIPTION:
XS GIS Cut Line= 3
      1636855.01      6923688.02      1637055.00      6924038.00
      1637404.99      6924787.97
#Sta/Elev= 30
  4632.2 1705.60  4677.5 1704.60  4758.1 1698.75  4816.5 1680.56  4838.8 1667.08
  4844.5 1666.39  4860.4 1660.65  4882.0 1655.89  4919.4 1652.05  4931.6 1649.11
  4954.7 1647.83  4977.7 1643.97  4988.1 1639.21  4988.7 1638.71  5011.8 1639.21
  5044.0 1644.38  5079.4 1646.52  5134.6 1645.66  5178.7 1648.32  5334.8 1650.57
  5357.7 1652.88  5375.0 1656.50  5426.3 1659.91  5500.3 1659.71  5631.2 1654.05
  5734.5 1660.32  5763.6 1664.48  5796.7 1666.30  5825.9 1671.12  5862.9 1674.36
#Mann=3,-1,0
  4632.2    0.05       0  4988.1    0.03       0  5011.8    0.05       0
Bank Sta=4988.1,5011.8
Exp/Cntr=0.3,0.1

Type RM Length L Ch R = 1,20448,655,655,655
BEGIN DESCRIPTION:
Long Creek 36.0
END DESCRIPTION:
XS GIS Cut Line= 3
      1636404.99      6924037.99      1636605.00      6924388.00
      1637355.00      6924988.00
#Sta/Elev= 30
  4634.3 1700.43  4707.0 1695.85  4744.5 1691.53  4818.6 1675.01  4830.8 1667.55
  4853.1 1659.22  4868.3 1655.53  4927.3 1648.28  4970.5 1639.04  4979.8 1638.97
  4986.3 1637.21  4988.2 1634.53  4989.2 1634.03  5027.7 1634.53  5029.5 1637.77
  5034.5 1641.34  5040.6 1641.34  5051.0 1644.16  5073.4 1645.65  5222.3 1647.70
  5414.4 1646.61  5649.7 1648.06  5670.5 1649.12  5769.8 1659.54  5784.2 1662.19
  5805.8 1669.68  5813.0 1670.81  5905.9 1676.31  5976.3 1678.58  5997.9 1680.78
#Mann=3,-1,0
  4634.3    0.05       0  4988.2    0.05       0  5027.7    0.05       0
Bank Sta=4988.2,5027.7
Exp/Cntr=0.3,0.1

Type RM Length L Ch R = 1,19793,422,422,422
BEGIN DESCRIPTION:
Long Creek 35.0
END DESCRIPTION:
XS GIS Cut Line= 3
      1635979.99      6924963.00      1636254.50      6924913.04
      1636904.15      6924743.61
#Sta/Elev= 30
  4714.5 1668.07  4767.8 1668.57  4821.2 1665.59  4851.7 1661.73  4872.1 1657.63
  4879.6 1654.76  4884.7 1654.71  4902.5 1650.87  4938.0 1647.34  4943.2 1645.30
  4983.9 1633.75  4984.6 1631.77  4985.6 1631.27  5023.2 1631.27  5024.2 1631.77
  5025.0 1633.48  5031.8 1637.35  5036.9 1637.06  5045.7 1641.75  5056.0 1643.53
  5077.4 1644.34  5087.0 1643.60  5107.6 1643.45  5159.4 1645.07  5183.6 1645.06
  5376.4 1646.74  5438.4 1645.85  5479.3 1646.01  5507.2 1645.50  5664.9 1646.08
#Mann=5,-1,0
  4714.5    0.05       0  4984.6    0.03       0  5024.2    0.05       0
  5183.6    0.12       0  5479.3    0.05       0
Bank Sta=4984.6,5024.2
Exp/Cntr=0.3,0.1
