HEC-RAS study South Prong Long Creek.prj: South Prong Long Creek Base Level Engineering

--- South Prong Long Creek.g01 (geometry) --- (continued)

Type RM Length L Ch R = 1,48990,270,270,270
BEGIN DESCRIPTION:
South Prong Long Creek 88.0
END DESCRIPTION:
XS GIS Cut Line= 3
      1656305.00      6897888.00      1656505.00      6898038.00
      1657399.02      6898240.65
#Sta/Elev= 30
  4739.1 1867.55  4775.6 1864.42  4781.8 1864.31  4796.4 1862.41  4817.2 1861.05
  4831.8 1859.31  4867.2 1853.84  4889.1 1851.97  4925.6 1850.51  4946.4 1850.94
  4952.6 1849.41  4976.1 1848.05  4976.6 1847.55  4987.1 1847.55  4987.6 1848.05
  5008.1 1849.28  5013.2 1851.08  5050.6 1855.05  5071.1 1855.98  5081.4 1855.25
  5112.1 1854.91  5214.7 1854.67  5266.0 1855.83  5296.7 1855.62  5409.5 1856.80
  5421.9 1856.50  5440.3 1857.04  5513.2 1857.03  5690.9 1858.82  5905.8 1862.15
#Mann=3,-1,0
  4739.1    0.05       0  4976.1    0.05       0  4987.6    0.05       0
Bank Sta=4976.1,4987.6
Exp/Cntr=0.3,0.1

Type RM Length L Ch R = 1,48720,176,176,176
BEGIN DESCRIPTION:
Mapping XS 6bd10311
END DESCRIPTION:
XS GIS Cut Line= 3
      1656180.27      6897990.61      1656258.41      6898152.11
      1656861.30      6898671.84
#Sta/Elev= 30
  4727.2 1869.74  4790.4 1866.66  4841.2 1861.26  4886.3 1858.56  4891.9 1857.29
  4906.6 1857.18  4936.9 1852.69  4951.1 1851.58  4957.7 1852.37  4965.4 1850.60
  4972.0 1851.82  4979.6 1850.46  5000.5 1851.74  5007.7 1851.52  5009.0 1850.46
  5009.5 1849.96  5020.6 1850.46  5021.4 1851.96  5029.0 1850.80  5035.6 1851.97
  5043.3 1851.20  5049.9 1852.22  5106.9 1852.83  5149.7 1850.64  5192.5 1851.92
  5199.1 1850.99  5213.3 1852.93  5219.9 1852.26  5248.5 1854.05  5702.6 1858.84
#Mann=3,-1,0
  4727.2    0.05       0  5009.0    0.03       0  5020.6    0.05       0
Bank Sta=5009,5020.6
Exp/Cntr=0.3,0.1

Type RM Length L Ch R = 1,48544,416,416,416
BEGIN DESCRIPTION:
South Prong Long Creek 87.0
END DESCRIPTION:
XS GIS Cut Line= 3
      1656054.97      6898237.98      1656205.00      6898338.00
      1657024.03      6899016.69
#Sta/Elev= 30
  4814.4 1865.90  4886.5 1860.28  4915.1 1858.90  4958.7 1852.25  4991.7 1849.05
  5031.2 1848.04  5031.7 1847.54  5042.9 1848.04  5051.4 1849.48  5059.2 1849.08
  5129.5 1852.08  5137.3 1850.86  5164.7 1849.27  5201.1 1850.24  5207.6 1851.47
  5215.5 1850.82  5222.0 1852.35  5228.5 1851.61  5242.8 1852.32  5300.1 1852.35
  5363.9 1853.86  5406.9 1853.53  5520.2 1855.64  5577.5 1855.47  5761.1 1858.22
  5769.0 1858.93  5775.5 1858.45  5783.3 1859.20  5989.1 1864.47  6058.4 1867.95
#Mann=3,-1,0
  4814.4    0.05       0  5031.2    0.03       0  5042.9    0.05       0
Bank Sta=5031.2,5042.9
Exp/Cntr=0.3,0.1

Type RM Length L Ch R = 1,48128,202,202,202
BEGIN DESCRIPTION:
South Prong Long Creek 86.0
END DESCRIPTION:
XS GIS Cut Line= 3
      1655855.03      6898538.03      1656005.00      6898688.00
      1656570.43      6898990.40
#Sta/Elev= 30
  4783.3 1862.44  4839.8 1859.45  4896.4 1857.33  4953.0 1850.90  4981.2 1848.55
  4991.8 1847.31  5009.2 1846.87  5047.4 1848.52  5085.6 1847.86  5101.4 1846.56
  5101.9 1846.06  5113.2 1846.06  5113.7 1846.56  5129.5 1848.69  5135.2 1848.52
  5142.8 1850.05  5157.1 1849.75  5165.5 1850.19  5217.3 1850.29  5343.3 1852.54
  5469.2 1853.68  5474.9 1853.28  5491.2 1853.93  5496.9 1853.55  5535.1 1854.34
  5540.7 1854.09  5573.3 1854.51  5595.2 1855.22  5622.8 1855.15  5636.6 1855.65
#Mann=3,-1,0
  4783.3    0.05       0  5101.4    0.03       0  5113.7    0.05       0
Bank Sta=5101.4,5113.7
Exp/Cntr=0.3,0.1

Type RM Length L Ch R = 1,47926,255,255,255
BEGIN DESCRIPTION:
Mapping XS 3f685c61
END DESCRIPTION:
XS GIS Cut Line= 2
      1655643.84      6898709.41      1656284.43      6899068.76
#Sta/Elev= 30
  4678.3 1862.38  4701.5 1861.50  4714.0 1860.68  4847.5 1856.08  4853.3 1855.45
  4863.1 1855.02  4874.9 1853.39  4885.2 1852.94  4890.9 1852.15  4920.4 1849.58
  4934.3 1848.77  4950.2 1848.46  4987.9 1846.90  4993.6 1845.89  5017.5 1843.80
  5018.0 1843.30  5029.3 1843.30  5029.8 1843.80  5031.2 1844.26  5037.0 1844.91
  5052.9 1845.41  5058.6 1846.48  5068.9 1846.91  5074.6 1848.14  5112.2 1849.22
  5126.8 1849.29  5199.0 1851.00  5252.6 1851.71  5274.3 1851.61  5412.8 1852.59
#Mann=3,-1,0
  4678.3    0.05       0  5017.5    0.03       0  5029.8    0.05       0
Bank Sta=5017.5,5029.8
Exp/Cntr=0.3,0.1

Type RM Length L Ch R = 1,47671,877,877,877
BEGIN DESCRIPTION:
South Prong Long Creek 85.0
END DESCRIPTION:
XS GIS Cut Line= 3
      1655554.99      6898837.99      1655755.00      6899038.00
      1656518.87      6899376.09
#Sta/Elev= 30
  4716.3 1860.85  4857.7 1855.09  4900.2 1851.91  4956.7 1848.78  4985.0 1845.77
  4989.5 1844.74  4990.0 1844.24  5001.3 1844.24  5001.8 1844.74  5021.0 1845.60
  5036.8 1845.07  5083.4 1848.16  5135.4 1847.70  5257.4 1850.32  5408.0 1851.67
  5431.3 1852.35  5545.9 1852.96  5553.2 1853.71  5558.7 1853.23  5582.0 1853.43
  5605.3 1854.06  5622.5 1853.94  5628.6 1854.47  5634.0 1854.01  5644.4 1854.51
  5657.3 1854.27  5666.2 1854.78  5710.0 1854.99  5825.8 1857.28  5834.5 1857.11
#Mann=3,-1,0
  4716.3    0.05       0  4989.5    0.03       0  5001.8    0.05       0
Bank Sta=4989.5,5001.8
Exp/Cntr=0.3,0.1

Type RM Length L Ch R = 1,46794,553,553,553
BEGIN DESCRIPTION:
South Prong Long Creek 84.0
END DESCRIPTION:
XS GIS Cut Line= 3
      1655190.69      6899027.08      1655605.00      6899638.00
      1655955.01      6900138.01
#Sta/Elev= 30
  4267.7 1859.94  4393.4 1856.78  4423.3 1855.04  4516.2 1851.82  4567.1 1848.18
  4595.0 1847.35  4681.0 1846.62  4716.9 1844.91  4740.0 1846.25  4776.3 1846.48
  4897.1 1845.83  4977.0 1842.40  4977.5 1841.90  4989.3 1841.90  4989.8 1842.40
  4998.4 1842.88  5002.8 1844.41  5008.9 1844.41  5028.1 1846.81  5069.9 1849.14
  5192.0 1849.67  5308.0 1851.29  5343.7 1852.55  5394.3 1855.64  5421.3 1858.41
  5451.0 1859.96  5465.8 1861.64  5486.7 1862.79  5573.0 1865.06  5616.2 1867.61
#Mann=3,-1,0
  4267.7    0.05       0  4977.0    0.03       0  4989.8    0.05       0
Bank Sta=4977,4989.8
Exp/Cntr=0.3,0.1

Type RM Length L Ch R = 1,46241,514,514,514
BEGIN DESCRIPTION:
South Prong Long Creek 83.0
END DESCRIPTION:
XS GIS Cut Line= 3
      1655034.46      6899136.53      1655138.62      6899610.44
      1655754.99      6900187.99
#Sta/Elev= 30
  4589.3 1857.71  4631.8 1856.79  4752.2 1852.04  4785.3 1851.39  4826.3 1849.83
  4893.7 1845.56  4928.7 1844.42  4937.5 1843.73  4942.6 1844.14  4949.2 1843.23
  4969.6 1841.92  4994.0 1841.16  4994.5 1840.66  5006.3 1840.66  5006.8 1841.16
  5035.3 1841.42  5070.7 1842.82  5105.7 1843.45  5140.8 1844.96  5176.5 1845.56
  5466.6 1846.36  5487.7 1846.83  5508.7 1846.56  5650.3 1848.48  5707.0 1850.45
  5735.3 1852.28  5784.6 1857.62  5806.1 1858.52  5855.5 1862.41  5919.2 1863.75
#Mann=3,-1,0
  4589.3    0.05       0  4994.0    0.03       0  5006.8    0.05       0
Bank Sta=4994,5006.8
Exp/Cntr=0.3,0.1

Type RM Length L Ch R = 1,45727,100,100,100
BEGIN DESCRIPTION:
South Prong Long Creek 82.0
END DESCRIPTION:
XS GIS Cut Line= 3
      1654724.89      6899534.90      1654830.00      6899863.00
      1655710.78      6900386.04
#Sta/Elev= 30
  4583.8 1846.35  4628.6 1845.78  4650.1 1846.52  4666.0 1846.06  4671.2 1846.97
  4698.1 1845.22  4703.3 1846.27  4730.2 1844.69  4762.4 1844.35  4776.1 1842.81
  4799.8 1843.94  4826.7 1844.07  4971.2 1840.85  4995.9 1839.51  4996.4 1839.01
  5008.3 1839.01  5008.8 1839.51  5051.0 1840.60  5073.7 1843.07  5088.1 1843.65
  5168.0 1843.13  5294.7 1844.94  5337.5 1844.94  5534.3 1848.20  5549.9 1848.93
  5585.4 1852.85  5635.6 1856.86  5736.9 1859.64  5805.1 1862.42  5952.7 1864.67
#Mann=3,-1,0
  4583.8    0.05       0  4995.9    0.03       0  5008.8    0.05       0
Bank Sta=4995.9,5008.8
Exp/Cntr=0.3,0.1

Type RM Length L Ch R = 1,45627,129,129,129
BEGIN DESCRIPTION:
Mapping XS 44582191
END DESCRIPTION:
XS GIS Cut Line= 2
      1654451.11      6899646.89      1655393.85      6900469.84
#Sta/Elev= 30
  4506.7 1844.08  4723.2 1843.52  4765.0 1842.76  4871.3 1843.30  4914.0 1842.31
  4971.1 1839.05  4971.6 1838.55  4984.1 1839.05  5006.1 1840.12  5028.0 1839.37
  5034.6 1840.06  5042.2 1839.55  5048.8 1840.49  5056.1 1839.84  5063.1 1840.55
  5105.8 1840.48  5112.4 1842.05  5140.9 1843.18  5304.2 1843.97  5367.8 1844.98
  5382.0 1846.07  5445.6 1847.06  5453.2 1847.79  5488.4 1848.01  5495.0 1847.20
  5509.2 1847.24  5531.1 1848.50  5537.7 1847.78  5566.2 1847.86  5758.1 1852.07
#Mann=3,-1,0
  4506.7    0.05       0  4971.1    0.03       0  4984.1    0.05       0
Bank Sta=4971.1,4984.1
Exp/Cntr=0.3,0.1

Type RM Length L Ch R = 1,45498,769,769,769
BEGIN DESCRIPTION:
South Prong Long Creek 81.0
END DESCRIPTION:
XS GIS Cut Line= 3
      1653820.93      6899271.92      1654774.04      6900100.03
      1655096.42      6900453.61
#Sta/Elev= 30
  3793.5 1854.90  4020.7 1849.87  4282.7 1841.95  4381.8 1841.70  4431.8 1843.39
  4466.9 1843.63  4714.8 1842.24  4892.4 1843.06  4956.0 1841.59  4978.0 1838.63
  4978.5 1838.13  4991.0 1838.63  5019.6 1839.47  5053.4 1841.56  5062.5 1840.88
  5069.3 1842.01  5083.5 1842.38  5090.9 1841.80  5097.7 1842.64  5105.1 1841.99
  5111.9 1842.90  5119.3 1842.30  5140.3 1842.83  5232.1 1842.38  5296.3 1843.84
  5366.6 1846.25  5416.6 1850.16  5465.9 1851.92  5508.5 1854.56  5534.6 1855.05
#Mann=3,-1,0
  3793.5    0.05       0  4978.0    0.03       0  4991.0    0.05       0
Bank Sta=4978,4991
Exp/Cntr=0.3,0.1

Type RM Length L Ch R = 1,44729,460,460,460
BEGIN DESCRIPTION:
South Prong Long Creek 80.0
END DESCRIPTION:
XS GIS Cut Line= 3
      1653837.39      6899414.23      1654158.58      6900460.27
      1654314.81      6900768.39
#Sta/Elev= 30
  3981.2 1850.86  4016.5 1850.54  4224.5 1844.98  4319.9 1842.25  4333.2 1841.22
  4365.9 1840.01  4398.6 1840.03  4414.0 1839.32  4436.6 1841.03  4455.9 1841.25
  4591.9 1840.22  4910.4 1840.21  4948.4 1839.38  4958.0 1838.55  4975.9 1835.60
  5002.1 1834.97  5002.6 1834.47  5014.6 1834.47  5015.1 1834.97  5041.3 1838.48
  5046.6 1838.45  5052.1 1839.85  5062.6 1840.72  5075.4 1841.19  5078.5 1841.79
  5100.8 1842.37  5139.7 1845.04  5241.1 1848.55  5398.0 1852.19  5420.9 1853.23
#Mann=3,-1,0
  3981.2    0.05       0  5002.1    0.03       0  5015.1    0.05       0
Bank Sta=5002.1,5015.1
Exp/Cntr=0.3,0.1

Type RM Length L Ch R = 1,44269,322,322,322
BEGIN DESCRIPTION:
South Prong Long Creek 79.0
END DESCRIPTION:
XS GIS Cut Line= 3
      1653455.00      6899188.00      1653676.86      6900387.55
      1653997.98      6900928.99
#Sta/Elev= 30
  3780.1 1861.34  3917.5 1857.50  3922.6 1857.86  4146.2 1850.17  4268.2 1847.42
  4329.3 1845.24  4400.4 1843.71  4481.8 1840.75  4519.9 1840.22  4532.7 1839.37
  4705.5 1837.44  4736.0 1838.67  4910.6 1839.11  4949.6 1836.88  4958.5 1834.36
  4983.7 1832.96  4984.2 1832.46  4996.3 1832.46  4996.8 1832.96  5006.2 1833.11
  5021.9 1837.75  5035.4 1838.63  5093.5 1838.91  5138.8 1840.40  5144.6 1840.10
  5181.7 1841.49  5187.5 1842.19  5209.8 1842.24  5458.4 1848.69  5629.5 1852.01
#Mann=3,-1,0
  3780.1    0.05       0  4983.7    0.03       0  4996.8    0.05       0
Bank Sta=4983.7,4996.8
Exp/Cntr=0.3,0.1

Type RM Length L Ch R = 1,43947,652,652,652
BEGIN DESCRIPTION:
South Prong Long Creek 78.0
END DESCRIPTION:
XS GIS Cut Line= 3
      1653054.99      6899587.97      1653355.00      6900388.00
      1653955.00      6901288.01
#Sta/Elev= 30
  4146.5 1855.53  4381.5 1848.61  4588.9 1841.05  4699.2 1836.00  4766.0 1835.66
  4814.9 1836.55  4851.4 1834.61  4875.4 1837.53  4936.8 1837.93  4979.6 1836.14
  4985.8 1834.88  4991.1 1835.08  5001.9 1832.43  5002.4 1831.93  5015.0 1832.43
  5023.5 1834.31  5029.5 1834.38  5044.5 1837.90  5059.5 1838.36  5173.7 1837.71
  5239.8 1836.46  5260.8 1835.12  5296.9 1835.75  5375.0 1840.13  5600.4 1845.02
  5794.1 1850.91  5966.9 1854.95  5974.4 1856.13  5987.9 1855.55  6082.6 1857.97
#Mann=3,-1,0
  4146.5    0.05       0  5001.9    0.05       0  5015.0    0.05       0
Bank Sta=5001.9,5015
Exp/Cntr=0.3,0.1

Type RM Length L Ch R = 1,43295,560,560,560
BEGIN DESCRIPTION:
South Prong Long Creek 77.0
END DESCRIPTION:
XS GIS Cut Line= 3
      1652639.51      6899956.84      1652911.08      6900385.80
      1653904.98      6901337.98
#Sta/Elev= 30
  4492.3 1845.53  4626.9 1843.93  4888.0 1838.92  4955.0 1836.21  4967.1 1833.41
  4982.1 1831.98  4990.8 1832.39  5018.8 1831.10  5019.3 1830.60  5031.7 1830.60
  5032.2 1831.10  5032.8 1831.72  5039.7 1833.24  5046.9 1834.20  5110.4 1835.44
  5223.7 1835.84  5343.8 1835.22  5407.3 1835.85  5435.6 1833.59  5471.2 1835.53
  5499.5 1836.31  5704.5 1839.02  5711.7 1839.76  5753.9 1840.30  5888.5 1843.98
  5902.6 1844.98  6001.7 1848.56  6192.6 1853.70  6249.2 1854.66  6376.4 1858.94
#Mann=3,-1,0
  4492.3    0.05       0  5018.8    0.05       0  5032.2    0.05       0
Bank Sta=5018.8,5032.2
Exp/Cntr=0.3,0.1

Type RM Length L Ch R = 1,42735,386,386,386
BEGIN DESCRIPTION:
Mapping XS 69447e92
END DESCRIPTION:
XS GIS Cut Line= 3
      1652405.07      6900317.52      1652513.62      6900746.73
      1653181.03      6901041.43
#Sta/Elev= 30
  4228.1 1836.65  4269.9 1835.60  4311.1 1835.18  4641.2 1832.65  4656.4 1832.90
  4668.9 1832.36  4682.1 1832.91  4687.5 1832.46  4770.7 1833.11  4891.0 1832.74
  4908.3 1831.25  4923.8 1830.69  4983.7 1831.22  4989.3 1829.98  5000.3 1828.52
  5000.8 1828.02  5013.2 1828.02  5013.7 1828.52  5022.1 1829.24  5035.7 1829.49
  5044.0 1830.67  5053.6 1831.34  5105.7 1833.70  5152.3 1833.74  5175.2 1832.84
  5197.0 1833.95  5233.1 1833.97  5308.5 1835.52  5339.2 1835.73  5400.4 1837.22
#Mann=3,-1,0
  4228.1    0.05       0  5000.3    0.03       0  5013.7    0.05       0
Bank Sta=5000.3,5013.7
Exp/Cntr=0.3,0.1

Type RM Length L Ch R = 1,42349,262,262,262
BEGIN DESCRIPTION:
Mapping XS 74ede5fc
END DESCRIPTION:
XS GIS Cut Line= 3
      1652391.39      6900347.11      1652422.47      6900764.09
      1652817.45      6901562.72
#Sta/Elev= 30
  4091.4 1836.08  4292.8 1833.20  4302.9 1833.59  4493.4 1831.72  4590.3 1831.30
  4657.6 1831.96  4915.5 1830.93  4977.3 1829.49  5005.3 1827.22  5009.2 1826.43
  5009.7 1825.93  5022.2 1825.93  5022.7 1826.43  5027.7 1827.16  5038.2 1827.14
  5050.2 1828.20  5060.6 1829.59  5067.0 1831.26  5072.6 1831.22  5089.4 1832.84
  5095.0 1832.57  5134.3 1834.49  5139.9 1834.31  5179.2 1837.14  5239.0 1838.41
  5246.5 1839.15  5252.1 1838.69  5319.4 1840.39  5328.3 1841.17  5400.5 1842.04
#Mann=3,-1,0
  4091.4    0.05       0  5009.2    0.03       0  5022.7    0.05       0
Bank Sta=5009.2,5022.7
Exp/Cntr=0.3,0.1

Type RM Length L Ch R = 1,42087,595,595,595
BEGIN DESCRIPTION:
South Prong Long Creek 76.0
END DESCRIPTION:
XS GIS Cut Line= 3
      1652326.98      6900594.77      1652405.00      6901188.00
      1652491.70      6901483.82
#Sta/Elev= 30
  4400.8 1832.51  4555.4 1831.13  4615.9 1831.28  4652.6 1830.62  4686.5 1830.87
  4716.7 1830.32  4827.7 1830.41  4928.5 1829.78  4948.7 1828.92  4957.3 1827.94
  4962.3 1828.36  4968.9 1827.36  4989.1 1826.09  5002.8 1824.70  5003.3 1824.20
  5015.8 1824.20  5016.3 1824.70  5030.4 1826.64  5049.3 1827.83  5054.5 1827.66
  5061.7 1829.17  5072.1 1830.40  5082.5 1831.02  5087.9 1831.98  5113.8 1833.02
  5154.7 1835.68  5193.3 1837.02  5249.2 1838.09  5304.0 1838.69  5307.4 1838.34
#Mann=3,-1,0
  4400.8    0.05       0  5002.8    0.05       0  5016.3    0.05       0
Bank Sta=5002.8,5016.3
Exp/Cntr=0.3,0.1

Type RM Length L Ch R = 1,41492,577,577,577
BEGIN DESCRIPTION:
Mapping XS c6c2dae3
END DESCRIPTION:
XS GIS Cut Line= 4
      1651957.89      6900209.14      1651923.34      6900642.56
      1651880.06      6901185.60      1652123.71      6901310.60
#Sta/Elev= 30
  4278.2 1837.72  4437.6 1834.48  4517.8 1832.07  4557.9 1831.50  4578.0 1830.80
  4588.0 1830.98  4658.3 1829.15  4754.3 1827.99  4768.6 1828.26  4778.6 1827.73
  4882.4 1827.51  4949.2 1826.16  4959.2 1825.23  4969.2 1823.78  4979.3 1823.20
  4998.8 1823.18  4999.3 1822.68  5011.9 1822.68  5012.4 1823.18  5039.5 1826.06
  5059.5 1826.70  5169.9 1827.50  5277.1 1827.08  5382.4 1828.93  5388.0 1828.70
  5404.6 1829.37  5471.2 1830.37  5476.9 1830.94  5493.4 1830.95  5531.6 1832.29
#Mann=3,-1,0
  4278.2    0.05       0  4998.8    0.05       0  5012.4    0.05       0
Bank Sta=4998.8,5012.4
Exp/Cntr=0.3,0.1

Type RM Length L Ch R = 1,40915,363,363,363
BEGIN DESCRIPTION:
Mapping XS 57628458
END DESCRIPTION:
XS GIS Cut Line= 3
      1651150.76      6900898.63      1651860.88      6901253.69
      1652055.19      6901332.18
#Sta/Elev= 30
  4743.6 1831.86  4887.8 1829.88  4893.7 1829.28  4910.2 1828.84  4926.9 1827.79
  4932.5 1828.00  4949.3 1825.83  4954.9 1825.65  4960.8 1823.88  4971.7 1822.13
  4977.3 1821.70  4983.1 1820.71  4987.2 1820.63  4987.7 1820.13  5000.4 1820.13
  5000.9 1820.63  5005.5 1821.78  5027.9 1822.84  5105.8 1824.61  5156.1 1824.32
  5178.5 1824.38  5184.4 1824.76  5206.7 1824.47  5245.6 1825.51  5379.8 1825.51
  5418.9 1826.23  5452.7 1825.81  5508.3 1825.98  5643.5 1828.15  5747.1 1830.41
#Mann=3,-1,0
  4743.6    0.05       0  4987.2    0.03       0  5000.9    0.05       0
Bank Sta=4987.2,5000.9
Exp/Cntr=0.3,0.1

Type RM Length L Ch R = 1,40552,133,133,133
BEGIN DESCRIPTION:
South Prong Long Creek 75.0
END DESCRIPTION:
XS GIS Cut Line= 3
      1650825.20      6901280.58      1651461.12      6901340.18
      1652170.38      6901397.74
#Sta/Elev= 30
  4361.3 1832.35  4501.7 1831.35  4521.8 1830.89  4541.9 1831.42  4708.2 1829.95
  4742.8 1830.11  4772.9 1829.47  4833.2 1829.03  4843.2 1828.44  4863.3 1828.44
  4903.5 1827.60  4913.5 1827.27  4943.6 1824.65  4983.8 1819.31  4987.0 1818.59
  4987.5 1818.09  5000.2 1818.09  5000.7 1818.59  5013.9 1819.34  5024.0 1820.89
  5031.9 1821.13  5036.9 1820.42  5054.1 1821.48  5064.1 1822.58  5124.3 1823.49
  5254.7 1823.76  5408.0 1826.11  5455.4 1827.52  5585.8 1830.25  5711.6 1833.69
#Mann=3,-1,0
  4361.3    0.05       0  4987.0    0.05       0  5000.7    0.05       0
Bank Sta=4987,5000.7
Exp/Cntr=0.3,0.1

Type RM Length L Ch R = 1,40419,1059,1059,1059
BEGIN DESCRIPTION:
South Prong Long Creek 74.0
END DESCRIPTION:
XS GIS Cut Line= 3
      1650807.90      6901423.81      1651504.94      6901458.57
      1652439.87      6901567.04
#Sta/Elev= 30
  4302.1 1832.73  4419.3 1831.10  4559.5 1830.00  4579.5 1829.39  4679.7 1829.46
  4749.8 1828.23  4769.8 1828.55  4849.9 1827.38  4891.5 1825.76  4940.0 1822.81
  4970.0 1819.33  4973.1 1818.31  4973.6 1817.81  4986.4 1817.81  4986.9 1818.31
  4990.0 1819.36  4997.5 1820.32  5010.1 1820.46  5030.3 1821.86  5312.1 1823.51
  5381.5 1825.37  5386.6 1825.06  5443.0 1827.30  5503.4 1828.70  5558.9 1830.85
  5563.9 1830.56  5604.1 1831.51  5664.5 1833.80  5814.9 1836.96  5941.2 1838.67
#Mann=3,-1,0
  4302.1    0.05       0  4973.1    0.03       0  4986.9    0.05       0
Bank Sta=4973.1,4986.9
Exp/Cntr=0.3,0.1

Type RM Length L Ch R = 1,39360,685,685,685
BEGIN DESCRIPTION:
South Prong Long Creek 73.0
END DESCRIPTION:
XS GIS Cut Line= 3
      1650555.02      6901638.01      1651755.00      6902338.00
      1652305.02      6902087.99
#Sta/Elev= 30
  3609.9 1837.72  3836.9 1831.95  4318.1 1823.68  4385.5 1823.40  4414.1 1822.65
  4420.3 1823.12  4457.1 1822.97  4478.6 1822.24  4515.8 1822.74  4524.5 1822.24
  4787.8 1819.02  4905.3 1818.57  4969.8 1816.55  4989.3 1813.91  4989.8 1813.41
  5002.7 1813.41  5003.2 1813.91  5013.4 1813.96  5031.0 1815.49  5036.5 1815.35
  5082.6 1822.00  5088.1 1821.51  5105.7 1823.01  5111.2 1822.80  5134.2 1824.11
  5226.5 1826.24  5255.1 1826.35  5317.7 1828.65  5375.9 1829.20  5603.3 1834.20
#Mann=3,-1,0
  3609.9    0.05       0  4989.3    0.05       0  5003.2    0.05       0
Bank Sta=4989.3,5003.2
Exp/Cntr=0.3,0.1

Type RM Length L Ch R = 1,38675,640,640,640
BEGIN DESCRIPTION:
Mapping XS 6f9800b5
END DESCRIPTION:
XS GIS Cut Line= 3
      1651033.49      6902702.45      1651617.88      6902981.57
      1651948.20      6902699.80
#Sta/Elev= 30
  4469.3 1820.83  4564.3 1819.12  4570.7 1818.67  4587.0 1818.62  4615.2 1817.62
  4648.3 1817.77  4677.7 1816.75  4683.2 1817.00  4751.3 1815.76  4825.6 1816.18
  4847.8 1815.92  4903.2 1816.56  4915.6 1816.33  4961.7 1813.33  4962.2 1812.83
  4975.1 1812.83  4975.6 1813.33  4983.7 1813.99  5000.8 1814.07  5046.2 1816.42
  5116.9 1816.03  5160.0 1816.27  5223.7 1817.37  5309.4 1817.58  5336.8 1818.07
  5358.8 1817.77  5415.5 1818.67  5422.5 1818.40  5514.7 1819.46  5551.1 1820.31
#Mann=3,-1,0
  4469.3    0.05       0  4961.7    0.05       0  4975.6    0.05       0
Bank Sta=4961.7,4975.6
Exp/Cntr=0.3,0.1

Type RM Length L Ch R = 1,38035,317,317,317
BEGIN DESCRIPTION:
South Prong Long Creek 72.0
END DESCRIPTION:
XS GIS Cut Line= 4
      1650751.42      6903389.96      1651155.00      6903338.00
      1651620.95      6902989.57      1651956.94      6902702.73
#Sta/Elev= 30
  4593.7 1829.10  4657.8 1827.80  4688.0 1826.74  4724.9 1824.78  4758.6 1823.93
  4809.5 1820.96  4883.9 1818.58  4919.9 1815.98  4930.0 1815.89  4970.4 1811.19
  4983.5 1810.44  4984.0 1809.94  4997.0 1809.94  4997.5 1810.44  5003.7 1810.70
  5022.5 1813.09  5072.5 1813.88  5314.3 1815.62  5472.7 1815.57  5572.7 1815.91
  5600.9 1816.43  5614.3 1816.11  5706.5 1817.57  5728.5 1817.32  5849.3 1817.91
  5870.1 1818.41  5884.4 1818.19  6005.2 1819.66  6019.4 1820.38  6024.2 1820.22
#Mann=3,-1,0
  4593.7    0.05       0  4983.5    0.03       0  4997.5    0.05       0
Bank Sta=4983.5,4997.5
Exp/Cntr=0.3,0.1

Type RM Length L Ch R = 1,37718,604,604,604
BEGIN DESCRIPTION:
Mapping XS f7277166
END DESCRIPTION:
XS GIS Cut Line= 3
      1651406.84      6903641.72      1651466.69      6903170.98
      1651876.63      6902783.09
#Sta/Elev= 30
  4794.7 1819.90  4821.7 1819.17  4828.7 1818.21  4848.9 1818.48  4896.6 1817.22
  4901.7 1817.40  4909.3 1816.93  4929.5 1815.38  4939.6 1813.89  4949.7 1812.30
  4959.7 1810.08  4962.8 1808.53  4963.3 1808.03  4976.4 1808.03  4976.9 1808.53
  5020.2 1809.04  5030.3 1809.94  5040.4 1811.67  5056.6 1812.79  5061.6 1812.58
  5136.5 1814.21  5277.3 1814.75  5291.5 1815.19  5319.8 1814.84  5425.8 1815.03
  5602.6 1816.96  5744.2 1817.55  5751.0 1817.94  5758.3 1817.70  5833.6 1818.36
#Mann=3,-1,0
  4794.7    0.05       0  4962.8    0.05       0  4976.9    0.05       0
Bank Sta=4962.8,4976.9
Exp/Cntr=0.3,0.1

Type RM Length L Ch R = 1,37114,73,73,73
BEGIN DESCRIPTION:
Mapping XS a8edb484
END DESCRIPTION:
XS GIS Cut Line= 5
      1651911.18      6903573.15      1651977.16      6903382.14
      1651987.58      6903284.92      1651959.80      6903177.28
      1651853.78      6902816.99
#Sta/Elev= 30
  4651.9 1819.64  4699.7 1817.90  4707.3 1817.91  4712.5 1818.50  4720.8 1817.30
  4816.0 1813.04  4826.6 1812.17  4832.0 1808.53  4837.3 1809.27  4853.5 1806.22
  4858.6 1806.22  4876.9 1804.05  4882.0 1804.82  4888.3 1803.65  4940.6 1803.39
  4941.1 1802.89  4954.2 1802.89  4954.7 1803.39  5051.9 1803.94  5098.2 1803.41
  5124.7 1807.46  5131.5 1808.93  5136.7 1807.93  5164.8 1811.14  5170.1 1810.75
  5176.8 1812.28  5187.3 1813.18  5203.4 1813.59  5208.6 1814.36  5438.5 1818.06
#Mann=3,-1,0
  4651.9    0.05       0  4940.6    0.05       0  4954.7    0.05       0
Bank Sta=4940.6,4954.7
Exp/Cntr=0.3,0.1

Type RM Length L Ch R = 1,37041,67,67,67
BEGIN DESCRIPTION:
Mapping XS 1d4f2cfa
END DESCRIPTION:
XS GIS Cut Line= 6
      1651963.26      6903562.75      1652046.61      6903323.12
      1652053.55      6903253.67      1652015.36      6903135.62
      1651958.36      6903045.94      1651898.09      6902802.84
#Sta/Elev= 30
  4657.6 1818.12  4789.7 1814.02  4790.4 1812.98  4790.9 1812.48  4804.5 1812.98
  4810.9 1817.22  4821.4 1817.08  4828.5 1815.29  4833.8 1817.60  4859.6 1817.08
  4864.9 1819.11  4890.7 1818.04  4916.5 1819.12  4943.5 1817.35  4948.5 1819.09
  4987.1 1819.08  4992.5 1818.80  4997.7 1815.99  5024.5 1817.88  5029.7 1813.70
  5056.5 1818.67  5061.7 1817.01  5093.8 1817.64  5111.7 1816.12  5117.6 1817.88
  5132.9 1816.28  5138.8 1818.31  5219.6 1817.79  5240.2 1813.58  5461.9 1818.01
#Mann=3,-1,0
  4657.6    0.05       0  4790.4    0.03       0  4804.5    0.05       0
Bank Sta=4790.4,4804.5
Exp/Cntr=0.3,0.1

Type RM Length L Ch R = 1,36974,702,702,702
BEGIN DESCRIPTION:
Mapping XS b3044e0b
END DESCRIPTION:
XS GIS Cut Line= 5
      1652036.17      6903580.09      1652126.47      6903402.98
      1652140.36      6903288.39      1652051.03      6903074.36
      1652188.42      6902887.35
#Sta/Elev= 30
  4585.1 1817.08  4698.8 1813.80  4733.4 1811.42  4778.3 1810.92  4783.9 1810.11
  4813.7 1809.06  4879.6 1809.22  4974.2 1807.22  4997.3 1807.40  5003.4 1808.24
  5027.2 1808.39  5032.6 1809.13  5051.0 1807.54  5056.5 1808.18  5073.2 1805.50
  5073.7 1805.00  5086.8 1805.00  5087.3 1805.50  5104.1 1806.44  5109.5 1805.91
  5126.6 1808.23  5139.1 1808.46  5152.1 1810.05  5160.5 1810.11  5166.7 1811.26
  5202.2 1813.44  5216.9 1811.97  5267.0 1814.65  5352.7 1816.12  5363.3 1815.86
#Mann=3,-1,0
  4585.1    0.05       0  5073.2    0.03       0  5087.3    0.05       0
Bank Sta=5073.2,5087.3
Exp/Cntr=0.3,0.1

Type RM Length L Ch R = 1,36272,508,508,508
BEGIN DESCRIPTION:
Mapping XS b80318c5
END DESCRIPTION:
XS GIS Cut Line= 2
      1652008.37      6903680.77      1653175.06      6903340.48
#Sta/Elev= 30
  4431.2 1817.19  4489.8 1814.98  4495.0 1815.35  4500.6 1814.63  4542.3 1813.80
  4562.0 1812.13  4567.2 1812.66  4600.7 1810.12  4605.9 1810.43  4646.4 1808.64
  4719.4 1807.94  4745.0 1808.27  4928.1 1805.79  4956.3 1803.59  4961.5 1803.67
  4969.4 1801.75  4982.5 1800.97  4983.0 1800.47  4996.6 1800.47  4997.1 1800.97
  5000.6 1802.54  5021.4 1807.17  5028.5 1807.51  5350.7 1809.53  5406.9 1811.52
  5500.6 1816.66  5567.2 1818.98  5583.9 1819.92  5600.7 1821.77  5646.5 1824.28
#Mann=3,-1,0
  4431.2    0.05       0  4982.5    0.03       0  4997.1    0.05       0
Bank Sta=4982.5,4997.1
Exp/Cntr=0.3,0.1

Type RM Length L Ch R = 1,35764,445,445,445
BEGIN DESCRIPTION:
South Prong Long Creek 71.0
END DESCRIPTION:
XS GIS Cut Line= 3
      1651938.27      6903772.70      1652455.00      6903988.00
      1653005.04      6903938.00
#Sta/Elev= 30
  4419.7 1817.04  4513.7 1812.30  4545.6 1811.57  4567.8 1808.62  4580.3 1807.92
  4657.2 1806.74  4947.0 1805.29  4957.8 1804.55  4964.9 1803.08  4970.3 1803.49
  4976.8 1802.22  4982.0 1802.22  4989.5 1800.74  4992.3 1798.99  4992.8 1798.49
  5006.9 1798.99  5019.7 1801.38  5059.8 1803.81  5089.9 1803.61  5150.2 1804.90
  5170.3 1804.49  5200.4 1802.33  5240.6 1803.66  5280.7 1808.37  5341.0 1812.10
  5361.1 1814.22  5401.2 1816.18  5411.3 1817.65  5471.5 1822.37  5531.8 1824.69
#Mann=3,-1,0
  4419.7    0.05       0  4992.3    0.03       0  5006.9    0.05       0
Bank Sta=4992.3,5006.9
Exp/Cntr=0.3,0.1

Type RM Length L Ch R = 1,35319,449,449,449
BEGIN DESCRIPTION:
South Prong Long Creek 70.0
END DESCRIPTION:
XS GIS Cut Line= 3
      1651804.99      6903787.99      1652355.00      6904338.00
      1652505.02      6904488.02
#Sta/Elev= 30
  4222.5 1820.10  4236.7 1819.10  4293.2 1817.10  4363.9 1813.48  4406.4 1812.06
  4448.8 1808.77  4477.1 1807.34  4561.9 1805.88  4689.2 1804.95  4774.1 1803.53
  4830.6 1803.48  4858.9 1802.46  4887.2 1802.08  4901.3 1800.55  4986.2 1799.69
  5021.2 1798.77  5021.7 1798.27  5035.6 1798.27  5036.1 1798.77  5042.8 1802.02
  5056.9 1804.17  5085.2 1806.63  5113.5 1808.52  5141.8 1811.31  5155.9 1813.87
  5170.0 1815.44  5177.1 1816.63  5184.2 1817.19  5208.9 1821.58  5212.5 1821.58
#Mann=3,-1,0
  4222.5    0.05       0  5021.2    0.05       0  5036.1    0.05       0
Bank Sta=5021.2,5036.1
Exp/Cntr=0.3,0.1

Type RM Length L Ch R = 1,34870,465,465,465
BEGIN DESCRIPTION:
South Prong Long Creek 69.0
END DESCRIPTION:
XS GIS Cut Line= 3
      1651505.03      6904088.03      1652105.00      6904688.00
      1652405.01      6904688.00
#Sta/Elev= 30
  4151.6 1817.21  4222.3 1815.40  4363.7 1810.23  4533.4 1806.46  4660.7 1804.40
  4703.1 1804.25  4717.2 1803.82  4802.1 1803.11  4816.2 1803.25  4858.7 1802.65
  4887.0 1802.79  4915.2 1802.16  4929.4 1801.57  4943.5 1799.60  4964.4 1796.08
  4964.9 1795.58  4978.8 1795.58  4979.3 1796.08  4996.6 1796.83  5020.1 1797.02
  5050.1 1798.94  5090.1 1799.99  5100.1 1800.85  5110.1 1802.29  5150.1 1805.84
  5170.1 1808.12  5200.1 1810.57  5250.1 1815.86  5280.1 1818.03  5300.1 1818.89
#Mann=3,-1,0
  4151.6    0.05       0  4964.4    0.05       0  4979.3    0.05       0
Bank Sta=4964.4,4979.3
Exp/Cntr=0.3,0.1

Type RM Length L Ch R = 1,34405,444,444,444
BEGIN DESCRIPTION:
South Prong Long Creek 68.0
END DESCRIPTION:
XS GIS Cut Line= 3
      1651305.00      6904538.00      1651905.00      6905088.00
      1652205.03      6905188.01
#Sta/Elev= 30
  4180.5 1814.06  4392.9 1806.31  4590.9 1802.19  4711.1 1800.45  4732.7 1800.61
  4753.6 1799.90  4775.2 1800.11  4782.0 1799.54  4789.4 1799.91  4803.6 1799.03
  4810.4 1799.70  4873.9 1800.48  4909.7 1800.67  4944.8 1800.04  4959.0 1799.43
  4973.2 1798.01  4980.6 1796.09  4987.3 1795.38  4991.0 1794.00  5008.0 1793.05
  5008.5 1792.55  5022.6 1792.55  5023.1 1793.05  5057.7 1795.78  5120.9 1803.61
  5194.7 1808.86  5215.8 1810.99  5236.9 1812.31  5289.6 1813.44  5310.7 1814.98
#Mann=3,-1,0
  4180.5    0.05       0  5008.0    0.05       0  5023.1    0.05       0
Bank Sta=5008,5023.1
Exp/Cntr=0.3,0.1

Type RM Length L Ch R = 1,33961,495,495,495
BEGIN DESCRIPTION:
South Prong Long Creek 67.0
END DESCRIPTION:
XS GIS Cut Line= 3
      1651234.10      6904896.02      1651655.00      6905438.00
      1652104.99      6906037.98
#Sta/Elev= 30
  4314.1 1812.35  4416.6 1808.25  4530.6 1801.03  4679.9 1798.33  4736.0 1796.52
  4779.5 1796.67  4835.7 1798.35  4928.8 1798.90  4978.6 1797.07  4986.8 1796.39
  4997.2 1794.26  5020.9 1792.19  5021.4 1791.69  5036.0 1792.19  5057.6 1792.40
  5072.2 1793.65  5093.0 1796.88  5113.9 1798.00  5213.9 1798.61  5322.2 1801.47
  5336.8 1802.45  5363.9 1806.40  5407.6 1808.84  5478.4 1815.24  5507.6 1816.49
  5550.3 1820.02  5578.4 1821.09  5607.6 1823.89  5686.8 1827.07  5750.3 1830.96
#Mann=3,-1,0
  4314.1    0.05       0  5020.9    0.05       0  5036.0    0.05       0
Bank Sta=5020.9,5036
Exp/Cntr=0.3,0.1

Type RM Length L Ch R = 1,33466,471,471,471
BEGIN DESCRIPTION:
South Prong Long Creek 66.0
END DESCRIPTION:
XS GIS Cut Line= 3
      1650904.99      6905387.99      1651305.00      6905788.00
      1651804.99      6906387.98
#Sta/Elev= 30
  4433.8 1814.82  4462.1 1813.01  4561.1 1809.83  4603.5 1807.59  4645.9 1803.70
  4674.2 1799.78  4702.5 1797.44  4744.9 1792.51  4759.1 1792.16  4801.5 1793.61
  4886.4 1793.77  5002.8 1792.12  5034.3 1790.11  5034.8 1789.61  5049.4 1790.11
  5049.6 1791.34  5056.1 1793.10  5077.6 1795.54  5134.2 1796.46  5233.8 1795.36
  5290.4 1796.93  5347.7 1800.16  5440.1 1809.61  5496.1 1812.80  5559.9 1819.75
  5602.8 1823.14  5680.9 1827.56  5702.4 1828.14  5759.0 1832.55  5780.5 1833.40
#Mann=3,-1,0
  4433.8    0.05       0  5034.3    0.03       0  5049.4    0.05       0
Bank Sta=5034.3,5049.4
Exp/Cntr=0.3,0.1

Type RM Length L Ch R = 1,32995,430,430,430
BEGIN DESCRIPTION:
South Prong Long Creek 65.0
END DESCRIPTION:
XS GIS Cut Line= 3
      1650855.00      6905537.98      1650905.00      6905788.00
      1651505.00      6906388.00
#Sta/Elev= 30
  4750.2 1809.08  4811.4 1805.72  4862.4 1799.38  4923.6 1793.61  4933.8 1791.68
  4944.0 1791.06  4977.1 1787.54  4977.6 1787.04  4992.0 1787.04  4992.5 1787.54
  5002.6 1788.70  5019.3 1788.76  5047.6 1790.13  5075.9 1790.48  5104.2 1791.99
  5146.6 1793.36  5231.4 1794.54  5316.3 1794.39  5471.9 1795.66  5514.3 1796.53
  5570.9 1798.58  5585.0 1799.17  5599.1 1802.09  5613.3 1803.39  5684.0 1805.63
  5712.3 1810.18  5740.6 1812.33  5768.8 1815.86  5811.3 1820.03  5853.7 1822.65
#Mann=3,-1,0
  4750.2    0.05       0  4977.1    0.03       0  4992.5    0.05       0
Bank Sta=4977.1,4992.5
Exp/Cntr=0.3,0.1

Type RM Length L Ch R = 1,32565,463,463,463
BEGIN DESCRIPTION:
South Prong Long Creek 64.0
END DESCRIPTION:
XS GIS Cut Line= 3
      1650555.00      6905638.02      1650505.00      6905888.00
      1651105.03      6906488.03
#Sta/Elev= 30
  4745.8 1805.33  4776.4 1803.92  4796.8 1802.33  4827.4 1798.09  4847.8 1796.03
  4888.6 1793.36  4929.3 1789.63  4949.7 1788.43  4970.1 1786.70  4990.5 1783.19
  4991.0 1782.69  5005.4 1782.69  5005.9 1783.19  5014.9 1783.39  5043.2 1788.79
  5057.3 1789.49  5142.2 1791.62  5311.9 1793.65  5354.3 1793.74  5396.7 1794.38
  5608.8 1795.94  5679.6 1797.65  5707.8 1799.03  5736.1 1801.42  5764.4 1804.75
  5806.8 1807.55  5821.0 1808.94  5835.1 1809.70  5845.7 1811.06  5849.3 1811.06
#Mann=3,-1,0
  4745.8    0.05       0  4990.5    0.03       0  5005.9    0.05       0
Bank Sta=4990.5,5005.9
Exp/Cntr=0.3,0.1

Type RM Length L Ch R = 1,32102,441,441,441
BEGIN DESCRIPTION:
South Prong Long Creek 63.0
END DESCRIPTION:
XS GIS Cut Line= 3
      1650005.00      6905738.01      1650055.00      6905938.00
      1650954.99      6906937.99
#Sta/Elev= 30
  4789.4 1807.81  4848.7 1806.32  4882.2 1803.52  4889.9 1802.18  4902.8 1798.02
  4913.1 1795.73  4936.3 1793.17  4944.0 1791.25  4964.6 1788.62  4985.2 1784.92
  4993.0 1782.92  4994.9 1780.75  4995.4 1780.25  5009.9 1780.25  5010.4 1780.75
  5031.1 1784.74  5037.8 1785.45  5073.7 1788.27  5094.6 1788.82  5200.7 1789.46
  5222.4 1789.07  5540.8 1792.83  5760.5 1797.36  5816.6 1799.25  5873.4 1802.13
  5930.2 1806.49  6015.4 1815.59  6135.7 1822.88  6319.6 1831.93  6340.9 1833.81
#Mann=3,-1,0
  4789.4    0.05       0  4994.9    0.03       0  5010.4    0.05       0
Bank Sta=4994.9,5010.4
Exp/Cntr=0.3,0.1

Type RM Length L Ch R = 1,31661,425,425,425
BEGIN DESCRIPTION:
South Prong Long Creek 62.0
END DESCRIPTION:
XS GIS Cut Line= 3
      1649655.00      6905987.99      1649705.00      6906188.00
      1650305.01      6906788.01
#Sta/Elev= 30
  4798.9 1805.33  4850.4 1800.84  4871.1 1796.17  4881.4 1794.84  4891.7 1792.84
  4904.6 1790.93  4912.3 1788.67  4932.9 1785.39  4945.8 1782.78  4953.5 1780.38
  4966.3 1779.30  4966.8 1778.80  4981.4 1778.80  4981.9 1779.30  4987.0 1780.53
  4994.8 1781.02  5008.6 1781.04  5019.2 1781.87  5047.5 1787.03  5104.1 1787.05
  5132.3 1786.64  5160.6 1786.89  5287.9 1789.89  5457.6 1791.66  5613.2 1794.59
  5726.3 1797.92  5782.9 1801.60  5825.3 1804.82  5850.1 1807.28  5853.6 1807.28
#Mann=3,-1,0
  4798.9    0.05       0  4966.3    0.03       0  4981.9    0.05       0
Bank Sta=4966.3,4981.9
Exp/Cntr=0.3,0.1

Type RM Length L Ch R = 1,31236,471,471,471
BEGIN DESCRIPTION:
South Prong Long Creek 61.0
END DESCRIPTION:
XS GIS Cut Line= 3
      1649405.00      6906087.98      1649355.00      6906388.00
      1649955.01      6906988.01
#Sta/Elev= 30
  4695.8 1802.55  4706.0 1802.39  4736.4 1800.82  4756.6 1798.24  4784.5 1793.38
  4789.6 1793.54  4797.2 1792.02  4817.5 1790.43  4845.4 1786.80  4850.4 1787.06
  4858.0 1786.34  4878.3 1785.49  4888.4 1783.60  4929.0 1782.57  4959.2 1780.68
  4959.7 1780.18  4974.3 1780.18  4974.8 1780.68  4989.8 1780.95  5056.5 1783.74
  5070.7 1783.52  5084.8 1783.83  5141.4 1786.87  5197.9 1787.30  5226.2 1786.93
  5282.8 1788.63  5523.2 1792.02  5650.5 1794.94  5763.6 1798.29  5848.5 1804.10
#Mann=3,-1,0
  4695.8    0.05       0  4959.2    0.03       0  4974.8    0.05       0
Bank Sta=4959.2,4974.8
Exp/Cntr=0.3,0.1

Type RM Length L Ch R = 1,30765,466,466,466
BEGIN DESCRIPTION:
South Prong Long Creek 60.0
END DESCRIPTION:
XS GIS Cut Line= 3
      1648805.01      6906288.03      1649005.00      6906688.00
      1649455.02      6907138.02
#Sta/Elev= 30
  4552.2 1804.07  4605.3 1799.91  4619.2 1797.61  4650.0 1791.31  4672.4 1787.91
  4694.7 1784.91  4717.1 1783.01  4761.8 1781.52  4798.1 1782.64  4865.2 1783.48
  4873.6 1783.06  4909.9 1782.76  4940.7 1780.92  4968.6 1780.48  4977.0 1779.50
  4985.4 1777.93  4988.7 1776.64  4989.2 1776.14  5003.9 1776.14  5004.4 1776.64
  5013.5 1776.81  5027.7 1779.16  5041.8 1782.59  5055.9 1783.74  5098.4 1785.52
  5154.9 1786.74  5169.1 1786.75  5197.4 1787.69  5296.4 1788.99  5635.8 1796.79
#Mann=3,-1,0
  4552.2    0.05       0  4988.7    0.03       0  5004.4    0.05       0
Bank Sta=4988.7,5004.4
Exp/Cntr=0.3,0.1

Type RM Length L Ch R = 1,30299,450,450,450
BEGIN DESCRIPTION:
South Prong Long Creek 59.0
END DESCRIPTION:
XS GIS Cut Line= 3
      1648555.00      6906488.01      1648555.00      6906738.00
      1649455.01      6907938.01
#Sta/Elev= 30
  4749.5 1798.80  4769.5 1797.23  4799.5 1791.37  4829.5 1787.05  4859.5 1781.06
  4869.5 1777.86  4879.5 1777.02  4899.5 1778.86  4939.5 1779.13  5002.6 1777.51
  5006.8 1776.06  5027.6 1776.31  5034.3 1775.52  5034.8 1775.02  5050.1 1775.52
  5056.8 1777.97  5077.6 1778.59  5085.9 1779.63  5092.2 1779.23  5099.5 1781.16
  5106.8 1781.91  5371.4 1785.43  5406.8 1785.00  5421.4 1786.19  5585.9 1789.18
  5842.2 1795.87  5963.0 1800.59  6135.9 1809.46  6363.0 1817.22  6499.5 1823.47
#Mann=3,-1,0
  4749.5    0.05       0  5034.3    0.03       0  5050.1    0.05       0
Bank Sta=5034.3,5050.1
Exp/Cntr=0.3,0.1

Type RM Length L Ch R = 1,29849,459,459,459
BEGIN DESCRIPTION:
South Prong Long Creek 58.0
END DESCRIPTION:
XS GIS Cut Line= 3
      1648004.98      6906637.98      1648155.00      6906788.00
      1649354.99      6907987.99
#Sta/Elev= 30
  4794.3 1797.89  4850.9 1795.10  4865.0 1793.88  4893.3 1788.10  4921.6 1783.81
  4949.9 1777.19  4964.0 1774.42  4984.3 1773.65  4984.8 1773.15  4999.8 1773.15
  5000.3 1773.65  5020.6 1774.91  5048.9 1775.73  5063.0 1777.88  5077.2 1778.94
  5091.3 1779.31  5162.0 1779.27  5459.0 1783.04  5487.3 1782.86  5529.7 1784.37
  5600.4 1785.09  5954.0 1793.49  6137.8 1800.79  6222.7 1804.90  6307.5 1808.19
  6335.8 1808.51  6420.7 1812.19  6505.5 1814.91  6604.5 1819.68  6703.5 1823.23
#Mann=3,-1,0
  4794.3    0.05       0  4984.3    0.05       0  5000.3    0.05       0
Bank Sta=4984.3,5000.3
Exp/Cntr=0.3,0.1

Type RM Length L Ch R = 1,29390,443,443,443
BEGIN DESCRIPTION:
South Prong Long Creek 57.0
END DESCRIPTION:
XS GIS Cut Line= 3
      1647604.97      6906837.97      1647755.00      6906988.00
      1648454.97      6907887.96
#Sta/Elev= 30
  4787.7 1793.15  4801.9 1791.73  4830.2 1786.71  4900.9 1781.41  4915.0 1779.59
  4929.2 1777.31  4943.3 1773.14  4963.5 1770.22  4964.0 1769.72  4979.6 1770.22
  5036.1 1775.79  5077.7 1777.50  5156.4 1777.38  5177.2 1776.50  5270.4 1777.75
  5291.2 1777.25  5448.7 1780.22  5463.2 1779.86  5527.4 1781.33  5548.2 1781.10
  5570.0 1782.08  5598.0 1781.89  5633.3 1783.55  5641.4 1782.99  5697.5 1784.39
  5755.5 1786.75  5875.8 1793.56  5904.8 1794.31  5933.7 1796.58  6140.0 1804.29
#Mann=3,-1,0
  4787.7    0.05       0  4963.5    0.05       0  4979.6    0.05       0
Bank Sta=4963.5,4979.6
Exp/Cntr=0.3,0.1

Type RM Length L Ch R = 1,28947,442,442,442
BEGIN DESCRIPTION:
South Prong Long Creek 56.0
END DESCRIPTION:
XS GIS Cut Line= 3
      1647405.00      6906887.98      1647405.00      6907188.00
      1648404.97      6907987.97
#Sta/Elev= 30
  4699.4 1792.84  4729.4 1790.53  4769.4 1786.12  4859.4 1779.84  4879.4 1777.55
  4919.4 1775.29  4959.4 1771.45  5033.7 1770.98  5034.2 1770.48  5049.4 1770.48
  5049.9 1770.98  5056.2 1772.60  5063.4 1773.19  5085.1 1774.55  5099.5 1774.82
  5205.1 1774.99  5383.6 1777.49  5533.3 1778.21  5690.2 1781.09  5696.6 1781.74
  5711.0 1781.68  5789.4 1784.06  5874.2 1789.80  5917.5 1791.60  5952.7 1794.06
  6010.3 1796.04  6037.5 1797.75  6202.4 1802.92  6223.2 1804.38  6280.0 1805.68
#Mann=3,-1,0
  4699.4    0.05       0  5033.7    0.03       0  5049.9    0.05       0
Bank Sta=5033.7,5049.9
Exp/Cntr=0.3,0.1

Type RM Length L Ch R = 1,28505,442,442,442
BEGIN DESCRIPTION:
South Prong Long Creek 55.0
END DESCRIPTION:
XS GIS Cut Line= 3
      1646954.99      6907237.98      1647055.00      6907438.00
      1647655.03      6908038.03
#Sta/Elev= 30
  4782.2 1790.47  4818.6 1787.56  4835.3 1785.87  4840.9 1784.82  4857.7 1783.75
  4863.3 1782.45  4880.0 1779.89  4908.0 1771.91  4916.4 1770.94  4924.8 1770.53
  4930.4 1771.02  5026.0 1770.24  5026.5 1769.74  5041.8 1769.74  5042.3 1770.24
  5076.5 1771.06  5090.7 1772.28  5175.5 1773.81  5189.7 1773.51  5288.7 1774.13
  5458.4 1774.31  5472.5 1774.74  5514.9 1774.41  5529.1 1774.98  5571.5 1774.78
  5670.5 1776.08  5755.4 1781.69  5826.1 1787.55  5850.8 1790.40  5854.4 1790.40
#Mann=3,-1,0
  4782.2    0.05       0  5026.0    0.03       0  5042.3    0.05       0
Bank Sta=5026,5042.3
Exp/Cntr=0.3,0.1

Type RM Length L Ch R = 1,28063,464,464,464
BEGIN DESCRIPTION:
South Prong Long Creek 54.0
END DESCRIPTION:
XS GIS Cut Line= 3
      1646554.99      6907688.00      1646755.00      6907738.00
      1647654.96      6908137.98
#Sta/Elev= 30
  4789.0 1790.37  4889.5 1786.03  4923.0 1783.64  4943.6 1778.39  4972.0 1773.44
  4977.1 1773.13  4992.6 1766.97  4997.9 1766.97  5001.4 1764.20  5001.9 1763.70
  5017.2 1763.70  5017.7 1764.20  5032.8 1765.09  5056.0 1769.22  5154.5 1771.14
  5214.0 1771.05  5268.7 1771.92  5450.0 1772.88  5487.6 1772.58  5640.8 1773.99
  5675.7 1775.14  5693.5 1775.07  5716.7 1775.85  5745.5 1778.45  5792.0 1780.39
  5826.8 1783.42  5837.8 1783.75  5903.4 1790.09  5947.9 1792.49  5980.0 1793.20
#Mann=3,-1,0
  4789.0    0.05       0  5001.4    0.05       0  5017.7    0.05       0
Bank Sta=5001.4,5017.7
Exp/Cntr=0.3,0.1

Type RM Length L Ch R = 1,27599,500,500,500
BEGIN DESCRIPTION:
South Prong Long Creek 53.0
END DESCRIPTION:
XS GIS Cut Line= 3
      1646504.96      6908087.98      1646705.00      6908188.00
      1647255.01      6908388.00
#Sta/Elev= 30
  4775.8 1784.26  4812.2 1781.73  4851.3 1776.45  4901.6 1771.39  4918.4 1766.89
  4940.8 1764.58  4946.3 1765.06  4963.1 1765.21  4977.1 1764.51  4985.5 1764.78
  4988.5 1763.70  4989.0 1763.20  5004.4 1763.20  5004.9 1763.70  5009.4 1765.21
  5031.4 1767.11  5040.0 1767.21  5045.3 1766.71  5101.2 1768.69  5126.5 1769.06
  5137.8 1768.57  5180.3 1769.69  5218.3 1769.47  5340.6 1770.24  5414.4 1771.81
  5446.4 1773.13  5467.6 1775.50  5531.5 1781.16  5569.4 1783.76  5584.7 1784.33
#Mann=3,-1,0
  4775.8    0.05       0  4988.5    0.03       0  5004.9    0.05       0
Bank Sta=4988.5,5004.9
Exp/Cntr=0.3,0.1

Type RM Length L Ch R = 1,27099,467,467,467
BEGIN DESCRIPTION:
South Prong Long Creek 52.0
END DESCRIPTION:
XS GIS Cut Line= 3
      1646255.01      6908438.00      1646705.00      6908688.00
      1647205.01      6908488.00
#Sta/Elev= 30
  4484.7 1790.10  4507.6 1789.02  4541.9 1785.58  4557.9 1785.07  4579.6 1782.72
  4617.4 1775.40  4667.7 1769.83  4704.3 1768.54  4770.7 1767.26  4793.6 1765.84
  4942.3 1764.63  4969.7 1762.67  4983.2 1760.56  4983.7 1760.06  4999.2 1760.06
  4999.7 1760.56  5002.2 1760.69  5008.9 1763.47  5014.3 1762.40  5021.0 1764.26
  5038.5 1766.18  5043.9 1765.74  5053.3 1766.86  5074.9 1767.91  5224.3 1769.77
  5236.4 1768.17  5268.7 1768.64  5445.1 1775.91  5469.3 1778.28  5538.0 1782.31
#Mann=3,-1,0
  4484.7    0.05       0  4983.2    0.05       0  4999.7    0.05       0
Bank Sta=4983.2,4999.7
Exp/Cntr=0.3,0.1

Type RM Length L Ch R = 1,26632,448,448,448
BEGIN DESCRIPTION:
South Prong Long Creek 51.0
END DESCRIPTION:
XS GIS Cut Line= 3
      1646104.98      6909088.00      1646505.00      6909088.00
      1647104.99      6909337.99
#Sta/Elev= 30
  4600.8 1780.75  4640.8 1776.78  4670.8 1773.03  4680.8 1772.29  4710.8 1768.95
  4720.8 1767.32  4730.8 1766.27  4770.8 1765.04  4830.8 1764.63  4850.8 1763.98
  4870.8 1763.86  4910.8 1762.03  4930.8 1762.16  4950.8 1761.08  4962.5 1759.38
  4963.0 1758.88  4978.6 1758.88  4979.1 1759.38  4980.8 1760.22  5015.4 1759.94
  5022.5 1760.87  5039.3 1762.15  5063.1 1763.31  5092.4 1763.33  5098.3 1763.75
  5121.6 1763.91  5239.1 1768.05  5390.8 1771.09  5535.4 1775.08  5650.8 1780.90
#Mann=3,-1,0
  4600.8    0.05       0  4962.5    0.03       0  4979.1    0.05       0
Bank Sta=4962.5,4979.1
Exp/Cntr=0.3,0.1

Type RM Length L Ch R = 1,26184,448,448,448
BEGIN DESCRIPTION:
South Prong Long Creek 50.0
END DESCRIPTION:
XS GIS Cut Line= 3
      1646054.97      6909237.97      1646355.00      6909488.00
      1646955.02      6909788.01
#Sta/Elev= 30
  4604.6 1780.57  4618.3 1779.77  4640.4 1777.22  4675.6 1774.92  4725.0 1769.82
  4732.9 1768.45  4739.4 1768.24  4747.2 1766.57  4753.7 1766.26  4768.0 1763.90
  4782.3 1763.07  4852.6 1762.09  4874.7 1762.59  4973.7 1761.80  4988.0 1760.67
  4991.9 1758.02  5009.1 1757.22  5048.3 1758.47  5070.6 1760.62  5093.0 1760.94
  5129.3 1758.44  5129.4 1757.09  5129.9 1756.59  5145.6 1756.59  5146.1 1757.09
  5160.1 1760.55  5188.0 1762.74  5218.8 1764.08  5584.9 1773.89  5666.0 1778.99
#Mann=3,-1,0
  4604.6    0.05       0  5129.4    0.03       0  5146.1    0.05       0
Bank Sta=5129.4,5146.1
Exp/Cntr=0.3,0.1

Type RM Length L Ch R = 1,25736,449,449,449
BEGIN DESCRIPTION:
South Prong Long Creek 49.0
END DESCRIPTION:
XS GIS Cut Line= 3
      1645854.99      6909738.00      1646355.00      6909938.00
      1646954.99      6909988.00
#Sta/Elev= 30
  4461.2 1776.94  4476.0 1776.10  4500.3 1773.53  4529.9 1772.42  4568.9 1769.43
  4601.2 1766.63  4608.0 1765.20  4613.3 1765.22  4622.8 1764.21  4859.7 1758.32
  4901.5 1759.23  4936.5 1758.83  4960.7 1758.02  4984.9 1755.99  5009.8 1755.13
  5011.4 1754.05  5011.9 1753.55  5027.6 1753.55  5028.1 1754.05  5029.8 1754.79
  5039.9 1755.31  5049.9 1756.52  5057.4 1758.75  5080.0 1760.74  5200.4 1765.28
  5303.3 1767.73  5401.1 1770.97  5441.3 1771.67  5501.5 1776.13  5601.8 1780.55
#Mann=3,-1,0
  4461.2    0.05       0  5011.4    0.05       0  5028.1    0.05       0
Bank Sta=5011.4,5028.1
Exp/Cntr=0.3,0.1

Type RM Length L Ch R = 1,25287,477,477,477
BEGIN DESCRIPTION:
South Prong Long Creek 48.0
END DESCRIPTION:
XS GIS Cut Line= 3
      1645873.03      6910190.31      1646205.00      6910338.00
      1646740.88      6910329.31
#Sta/Elev= 30
  4637.4 1768.83  4644.5 1768.87  4650.5 1767.36  4667.8 1765.29  4673.2 1765.56
  4683.3 1764.33  4691.0 1764.11  4705.2 1762.18  4727.1 1760.73  4737.5 1760.96
  4749.0 1760.07  4789.5 1758.95  4902.2 1756.67  4916.6 1755.76  4957.0 1754.51
  4968.6 1753.17  4978.9 1752.65  5012.3 1751.52  5012.8 1751.02  5028.6 1751.02
  5029.1 1751.52  5030.7 1752.18  5050.8 1754.54  5060.8 1756.46  5110.8 1760.14
  5190.8 1762.39  5440.8 1765.87  5500.8 1767.16  5520.8 1767.07  5536.7 1767.73
#Mann=3,-1,0
  4637.4    0.05       0  5012.3    0.03       0  5029.1    0.05       0
Bank Sta=5012.3,5029.1
Exp/Cntr=0.3,0.1

Type RM Length L Ch R = 1,24810,471,471,471
BEGIN DESCRIPTION:
South Prong Long Creek 47.0
END DESCRIPTION:
XS GIS Cut Line= 3
      1645904.98      6910738.00      1646105.00      6910738.00
      1647005.01      6910237.99
#Sta/Elev= 30
  4800.9 1777.56  4840.9 1773.65  4860.9 1768.60  4880.9 1764.54  4900.9 1762.31
  4910.9 1759.96  4920.9 1759.13  4940.9 1756.18  4960.9 1749.43  4962.5 1747.63
  4963.0 1747.13  4978.8 1747.13  4979.3 1747.63  4990.9 1748.75  5003.8 1748.81
  5014.7 1749.99  5030.7 1753.26  5068.4 1755.39  5103.9 1755.49  5111.9 1755.02
  5139.3 1756.06  5383.0 1761.40  5561.5 1763.67  5721.6 1766.50  5751.4 1767.81
  5767.4 1767.89  5838.3 1771.29  5881.8 1774.16  5995.0 1778.87  6030.5 1781.01
#Mann=3,-1,0
  4800.9    0.05       0  4962.5    0.05       0  4979.3    0.05       0
Bank Sta=4962.5,4979.3
Exp/Cntr=0.3,0.1

Type RM Length L Ch R = 1,24339,471,471,471
BEGIN DESCRIPTION:
South Prong Long Creek 46.0
END DESCRIPTION:
XS GIS Cut Line= 3
      1646255.03      6911237.97      1646405.00      6911088.00
      1646954.98      6910488.03
#Sta/Elev= 30
  4793.2 1775.01  4835.6 1772.06  4878.0 1765.02  4906.3 1761.33  4934.6 1756.36
  4962.9 1745.21  4982.7 1744.26  4983.2 1743.76  4999.1 1743.76  4999.6 1744.26
  5001.8 1745.95  5008.7 1745.95  5012.4 1747.71  5019.2 1749.84  5026.6 1751.04
  5033.4 1751.46  5090.1 1751.49  5097.5 1752.21  5104.3 1751.88  5203.5 1755.69
  5295.4 1757.84  5302.8 1757.54  5330.9 1758.66  5429.8 1760.08  5521.7 1762.08
  5578.4 1762.66  5649.4 1764.16  5783.8 1768.16  5805.4 1769.40  5819.2 1769.66
#Mann=3,-1,0
  4793.2    0.05       0  4982.7    0.03       0  4999.6    0.05       0
Bank Sta=4982.7,4999.6
Exp/Cntr=0.3,0.1

Type RM Length L Ch R = 1,23868,415,415,415
BEGIN DESCRIPTION:
South Prong Long Creek 45.0
END DESCRIPTION:
XS GIS Cut Line= 3
      1646504.98      6911488.00      1646705.00      6911438.00
      1647904.99      6910838.01
#Sta/Elev= 30
  4787.6 1772.89  4828.8 1770.91  4893.3 1762.35  4921.6 1760.61  4942.2 1757.39
  4962.8 1755.51  4975.7 1751.10  4991.2 1748.32  5002.2 1747.37  5024.5 1746.15
  5091.6 1746.98  5136.3 1745.65  5158.7 1744.79  5172.6 1741.63  5173.1 1741.13
  5189.5 1741.63  5195.0 1744.19  5203.4 1744.87  5209.0 1746.67  5231.4 1748.96
  5253.7 1750.44  5343.2 1753.06  5463.3 1754.27  5656.2 1753.09  5687.0 1751.81
  5740.1 1754.20  5843.5 1757.03  5969.3 1763.48  6209.6 1782.10  6335.4 1786.97
#Mann=3,-1,0
  4787.6    0.05       0  5172.6    0.05       0  5189.5    0.05       0
Bank Sta=5172.6,5189.5
Exp/Cntr=0.3,0.1

Type RM Length L Ch R = 1,23453,354,354,354
BEGIN DESCRIPTION:
South Prong Long Creek 44.0
END DESCRIPTION:
XS GIS Cut Line= 3
      1646504.96      6911838.01      1647055.00      6911638.00
      1647655.00      6911038.00
#Sta/Elev= 30
  4416.9 1764.31  4432.2 1764.55  4457.5 1763.13  4488.1 1763.43  4518.7 1762.49
  4544.0 1762.27  4549.3 1763.02  4605.1 1761.35  4610.5 1761.94  4635.7 1760.67
  4666.3 1760.84  4800.0 1758.33  4808.7 1757.92  4839.2 1753.48  4869.8 1752.39
  4875.2 1751.48  4925.7 1748.75  4931.0 1747.11  4961.6 1744.79  5030.5 1743.03
  5036.2 1741.91  5036.7 1741.41  5053.1 1741.91  5129.5 1742.97  5214.3 1748.37
  5327.4 1750.15  5454.7 1749.77  5638.6 1753.61  5780.0 1760.81  5850.7 1767.04
#Mann=3,-1,0
  4416.9    0.05       0  5036.2    0.05       0  5053.1    0.05       0
Bank Sta=5036.2,5053.1
Exp/Cntr=0.3,0.1
