HEC-RAS study Spring Creek.prj: Spring Creek Base Level Engineering

--- Spring Creek.g01 (geometry) --- (continued)

Type RM Length L Ch R = 1,83988,240,240,240
BEGIN DESCRIPTION:
Spring Creek 138.0
END DESCRIPTION:
XS GIS Cut Line= 3
      1660368.90      6875924.99      1660855.00      6876538.00
      1661355.03      6876938.02
#Sta/Elev= 30
  4217.7 1905.19  4238.1 1905.14  4345.5 1901.55  4502.3 1898.02  4566.1 1895.12
  4643.5 1892.90  4771.7 1893.47  4800.5 1891.35  4872.4 1891.95  4879.1 1891.33
  4907.9 1891.34  4943.2 1888.87  4949.5 1889.41  4964.0 1888.29  4972.0 1886.84
  4980.0 1886.70  4980.5 1886.20  4992.5 1886.20  4993.0 1886.70  4996.9 1888.92
  5007.3 1888.71  5013.7 1893.15  5021.7 1891.80  5028.1 1893.65  5092.1 1893.27
  5128.1 1894.09  5263.4 1902.72  5341.8 1905.37  5469.9 1911.38  5640.4 1923.60
#Mann=3,-1,0
  4217.7    0.05       0  4980.0    0.03       0  4993.0    0.05       0
Bank Sta=4980,4993
Exp/Cntr=0.3,0.1

Type RM Length L Ch R = 1,83748,574,574,574
BEGIN DESCRIPTION:
Mapping XS f017b19b
END DESCRIPTION:
XS GIS Cut Line= 2
      1660230.04      6876213.21      1661045.99      6876945.83
#Sta/Elev= 30
  4469.3 1898.89  4561.1 1897.45  4596.9 1897.41  4787.6 1892.57  4809.2 1891.19
  4830.2 1890.63  4858.6 1890.95  4915.4 1893.07  4936.3 1893.08  4943.8 1892.71
  4950.5 1889.19  4958.0 1887.20  4958.2 1886.69  4958.7 1886.19  4970.7 1886.19
  4971.2 1886.69  4986.4 1887.18  4993.1 1888.38  5014.1 1889.59  5056.7 1890.39
  5106.8 1892.11  5162.8 1891.67  5198.7 1892.17  5255.5 1890.85  5269.0 1891.19
  5290.6 1892.78  5361.7 1900.15  5375.9 1901.18  5467.8 1905.33  5565.9 1908.89
#Mann=3,-1,0
  4469.3    0.05       0  4958.2    0.03       0  4971.2    0.05       0
Bank Sta=4958.2,4971.2
Exp/Cntr=0.3,0.1

Type RM Length L Ch R = 1,83174,355,355,355
BEGIN DESCRIPTION:
Mapping XS f9f9417b
END DESCRIPTION:
XS GIS Cut Line= 3
      1659735.02      6876572.30      1660071.24      6876668.62
      1660806.42      6877261.81
#Sta/Elev= 30
  4006.4 1899.81  4155.7 1896.50  4189.5 1895.08  4223.2 1894.62  4228.4 1895.73
  4256.0 1894.32  4267.4 1894.69  4328.8 1891.22  4355.5 1888.86  4414.8 1886.95
  4429.2 1887.14  4458.0 1889.35  4493.2 1888.52  4542.8 1888.48  4571.6 1888.89
  4656.5 1891.77  4785.0 1892.13  4941.0 1890.18  4977.7 1887.66  5006.4 1884.82
  5006.9 1884.32  5019.0 1884.32  5019.5 1884.82  5033.8 1886.76  5048.2 1889.51
  5054.8 1891.76  5076.9 1895.30  5119.1 1898.49  5169.7 1900.89  5300.8 1905.04
#Mann=3,-1,0
  4006.4    0.05       0  5006.4    0.05       0  5019.5    0.05       0
Bank Sta=5006.4,5019.5
Exp/Cntr=0.3,0.1

Type RM Length L Ch R = 1,82819,875,875,875
BEGIN DESCRIPTION:
Mapping XS b4cd40bb
END DESCRIPTION:
XS GIS Cut Line= 4
      1659598.07      6876799.98      1659896.67      6876824.28
      1660355.00      6877317.34      1660590.51      6877383.15
#Sta/Elev= 30
  4067.8 1902.15  4205.2 1897.13  4224.3 1896.67  4235.3 1897.81  4275.4 1896.88
  4305.5 1895.10  4351.1 1896.78  4356.1 1895.60  4390.0 1893.35  4439.8 1885.77
  4475.0 1881.57  4482.6 1881.51  4483.1 1881.01  4495.7 1881.51  4524.3 1884.09
  4574.2 1885.80  4609.3 1887.96  4637.7 1888.34  4878.1 1888.06  4892.2 1887.80
  4913.7 1885.03  4927.9 1884.18  4970.4 1884.03  4991.4 1885.18  4998.8 1887.74
  5005.6 1887.26  5012.9 1889.54  5037.6 1893.04  5092.5 1893.58  5285.1 1898.48
#Mann=3,-1,0
  4067.8    0.05       0  4482.6    0.03       0  4495.7    0.05       0
Bank Sta=4482.6,4495.7
Exp/Cntr=0.3,0.1

Type RM Length L Ch R = 1,81944,68,68,68
BEGIN DESCRIPTION:
Mapping XS 09e11bc2
END DESCRIPTION:
XS GIS Cut Line= 6
      1659469.57      6877244.42      1659823.75      6877240.95
      1659920.97      6877150.67      1660080.69      6877258.31
      1660198.75      6877317.34      1660590.60      6877404.03
#Sta/Elev= 30
  4715.2 1903.82  4920.6 1893.49  4970.6 1880.53  4993.8 1878.18  4994.3 1877.68
  5007.5 1878.18  5114.7 1880.34  5171.4 1890.24  5218.5 1888.51  5245.6 1891.76
  5254.5 1890.66  5260.6 1893.08  5275.5 1889.69  5296.5 1891.32  5311.5 1888.49
  5332.5 1891.02  5362.5 1889.14  5368.5 1891.11  5405.1 1888.65  5410.7 1891.12
  5427.5 1889.32  5433.1 1891.05  5494.6 1889.68  5521.8 1892.48  5550.7 1891.44
  5555.8 1893.68  5594.3 1892.80  5599.4 1894.85  5625.2 1891.35  5928.0 1898.77
#Mann=3,-1,0
  4715.2    0.05       0  4993.8    0.05       0  5007.5    0.05       0
Bank Sta=4993.8,5007.5
Exp/Cntr=0.3,0.1

Type RM Length L Ch R = 1,81876,69,69,69
BEGIN DESCRIPTION:
Mapping XS decdf798
END DESCRIPTION:
XS GIS Cut Line= 6
      1659455.66      6877317.34      1659730.00      6877306.92
      1659872.36      6877324.28      1659952.22      6877220.12
      1660045.97      6877289.56      1660531.08      6877452.42
#Sta/Elev= 30
  4700.9 1903.27  4850.4 1894.91  5020.7 1896.89  5025.7 1892.65  5101.4 1895.83
  5117.7 1890.12  5139.4 1896.84  5225.7 1897.34  5257.4 1896.91  5292.8 1889.81
  5301.2 1893.47  5307.5 1890.32  5322.1 1896.22  5328.3 1891.99  5336.7 1895.69
  5342.9 1891.64  5351.3 1894.35  5357.6 1890.27  5374.3 1894.85  5379.6 1890.37
  5406.0 1896.43  5411.2 1892.58  5437.6 1896.33  5442.9 1893.59  5532.5 1896.42
  5595.5 1895.36  5625.4 1889.62  5625.9 1889.12  5639.1 1889.62  5878.5 1896.91
#Mann=3,-1,0
  4700.9    0.05       0  5625.4    0.03       0  5639.1    0.05       0
Bank Sta=5625.4,5639.1
Exp/Cntr=0.3,0.1

Type RM Length L Ch R = 1,81807,209,209,209
BEGIN DESCRIPTION:
Mapping XS 355eb765
END DESCRIPTION:
XS GIS Cut Line= 4
      1659549.40      6877359.00      1659830.69      6877386.78
      1660056.39      6877376.37      1660464.15      6877483.49
#Sta/Elev= 30
  4794.0 1898.90  4819.7 1896.21  4900.1 1893.13  4910.2 1891.14  4935.8 1884.48
  4940.9 1885.04  4983.7 1880.52  4984.2 1880.02  4996.9 1880.02  4997.4 1880.52
  5020.7 1880.71  5037.0 1883.00  5042.0 1882.26  5060.9 1882.90  5070.9 1884.51
  5076.3 1886.36  5101.0 1887.11  5121.0 1887.38  5171.1 1886.53  5181.1 1885.99
  5191.1 1883.16  5201.1 1883.82  5221.1 1887.17  5368.2 1889.91  5466.6 1891.27
  5489.3 1890.82  5605.2 1892.58  5640.4 1893.92  5645.5 1893.53  5724.2 1895.31
#Mann=3,-1,0
  4794.0    0.05       0  4983.7    0.03       0  4997.4    0.05       0
Bank Sta=4983.7,4997.4
Exp/Cntr=0.3,0.1

Type RM Length L Ch R = 1,81598,500,500,500
BEGIN DESCRIPTION:
Spring Creek 136.0
END DESCRIPTION:
XS GIS Cut Line= 3
      1659504.99      6877387.99      1659755.00      6877588.00
      1660955.03      6877588.00
#Sta/Elev= 30
  4680.5 1899.86  4772.6 1896.59  4830.2 1893.44  4836.6 1893.86  4844.6 1892.54
  4865.4 1891.33  4879.8 1887.97  4894.2 1886.72  4979.1 1882.41  4987.1 1881.00
  4993.5 1880.87  4997.5 1879.23  5013.8 1878.65  5014.3 1878.15  5027.5 1878.65
  5040.7 1879.52  5050.7 1881.22  5070.7 1881.31  5100.7 1885.64  5130.7 1884.99
  5140.7 1883.32  5150.7 1879.77  5160.7 1879.84  5190.7 1884.84  5230.7 1886.25
  5460.7 1891.03  5650.7 1893.79  5800.7 1897.66  6030.7 1907.07  6200.7 1919.86
#Mann=3,-1,0
  4680.5    0.05       0  5013.8    0.03       0  5027.5    0.05       0
Bank Sta=5013.8,5027.5
Exp/Cntr=0.3,0.1

Type RM Length L Ch R = 1,81098,464,464,464
BEGIN DESCRIPTION:
Spring Creek 135.0
END DESCRIPTION:
XS GIS Cut Line= 3
      1659505.01      6878038.00      1659755.00      6878088.00
      1660955.04      6877687.99
#Sta/Elev= 30
  4745.4 1899.50  4816.8 1896.85  4847.4 1894.07  4888.2 1888.18  4949.4 1883.40
  4979.9 1878.48  4997.8 1879.29  5032.0 1879.44  5042.5 1878.24  5046.1 1877.26
  5046.6 1876.76  5059.5 1876.76  5060.0 1877.26  5084.7 1878.56  5105.8 1882.12
  5116.3 1882.48  5158.5 1883.51  5200.6 1883.34  5242.8 1884.80  5422.0 1888.72
  5601.2 1891.62  5653.9 1893.39  5664.4 1893.11  5706.6 1894.46  5748.8 1894.94
  5822.5 1897.23  5927.9 1902.33  6043.9 1905.88  6096.6 1908.18  6265.3 1920.49
#Mann=3,-1,0
  4745.4    0.05       0  5046.1    0.03       0  5060.0    0.05       0
Bank Sta=5046.1,5060
Exp/Cntr=0.3,0.1

Type RM Length L Ch R = 1,80634,501,501,501
BEGIN DESCRIPTION:
Spring Creek 134.0
END DESCRIPTION:
XS GIS Cut Line= 3
      1659304.97      6878488.00      1659805.00      6878538.00
      1660535.52      6878254.85
#Sta/Elev= 30
  4503.7 1899.92  4564.0 1896.68  4644.4 1890.82  4664.5 1888.49  4825.3 1882.68
  4895.7 1880.90  4915.8 1877.21  4925.8 1876.77  4939.0 1875.14  4939.5 1874.64
  4952.4 1874.64  4952.9 1875.14  4953.5 1875.81  4966.0 1876.27  4996.2 1875.86
  5003.7 1876.56  5038.4 1876.94  5045.7 1878.54  5059.8 1878.93  5135.5 1880.13
  5154.7 1882.03  5274.4 1883.10  5432.5 1888.24  5516.9 1888.90  5531.7 1887.93
  5585.4 1889.53  5625.9 1889.37  5710.3 1890.43  5764.7 1891.61  5789.7 1892.85
#Mann=3,-1,0
  4503.7    0.05       0  4939.0    0.05       0  4952.9    0.05       0
Bank Sta=4939,4952.9
Exp/Cntr=0.3,0.1

Type RM Length L Ch R = 1,80133,447,447,447
BEGIN DESCRIPTION:
Spring Creek 133.0
END DESCRIPTION:
XS GIS Cut Line= 3
      1659454.99      6879088.00      1659805.00      6879038.00
      1660205.04      6879038.00
#Sta/Elev= 30
  4646.4 1887.33  4727.2 1884.22  4747.4 1882.97  4757.5 1881.56  4797.9 1879.41
  4828.2 1876.48  4858.5 1874.63  4868.6 1874.30  4878.7 1874.77  4898.9 1876.71
  4949.5 1877.09  4969.7 1876.73  4990.1 1866.78  4990.6 1866.28  5004.3 1866.28
  5004.8 1866.78  5010.0 1867.17  5020.0 1870.01  5030.0 1871.94  5050.0 1872.92
  5060.0 1874.12  5080.0 1879.17  5090.0 1880.03  5100.0 1877.96  5150.0 1881.61
  5260.0 1884.18  5270.0 1884.10  5330.0 1885.82  5380.0 1886.61  5400.0 1887.72
#Mann=3,-1,0
  4646.4    0.05       0  4990.1    0.05       0  5004.8    0.05       0
Bank Sta=4990.1,5004.8
Exp/Cntr=0.3,0.1

Type RM Length L Ch R = 1,79686,452,452,452
BEGIN DESCRIPTION:
Spring Creek 132.0
END DESCRIPTION:
XS GIS Cut Line= 3
      1659305.01      6879288.00      1659755.00      6879438.00
      1660254.97      6879537.99
#Sta/Elev= 30
  4520.5 1890.57  4615.4 1887.93  4741.8 1883.48  4794.6 1880.64  4847.3 1876.58
  4878.9 1874.92  4921.0 1871.58  4942.1 1871.17  4973.7 1871.39  4997.4 1870.47
  5005.0 1869.32  5015.2 1866.57  5018.1 1864.51  5018.6 1864.01  5032.3 1864.01
  5032.8 1864.51  5035.6 1864.94  5045.8 1868.28  5056.0 1870.88  5066.2 1871.53
  5086.6 1874.98  5158.0 1877.58  5178.4 1878.94  5290.6 1881.82  5331.4 1883.52
  5372.2 1886.13  5382.4 1887.32  5423.1 1889.60  5484.3 1895.16  5504.7 1896.12
#Mann=3,-1,0
  4520.5    0.05       0  5018.1    0.03       0  5032.8    0.05       0
Bank Sta=5018.1,5032.8
Exp/Cntr=0.3,0.1

Type RM Length L Ch R = 1,79234,466,466,466
BEGIN DESCRIPTION:
Spring Creek 131.0
END DESCRIPTION:
XS GIS Cut Line= 3
      1659355.03      6879788.01      1659605.00      6879838.00
      1660205.01      6879688.00
#Sta/Elev= 30
  4744.4 1883.06  4846.4 1880.63  4876.9 1879.34  4938.1 1875.08  4968.7 1872.36
  4978.9 1870.72  4989.1 1866.10  4989.4 1863.00  4989.9 1862.50  5003.7 1862.50
  5004.2 1863.00  5009.6 1863.96  5017.4 1866.43  5022.5 1866.27  5040.6 1867.84
  5063.7 1868.71  5092.1 1871.06  5246.7 1875.70  5277.6 1877.26  5360.1 1878.55
  5434.8 1880.56  5504.4 1883.74  5512.1 1884.40  5517.3 1884.32  5535.3 1886.68
  5545.6 1887.46  5553.4 1888.68  5558.5 1888.81  5566.2 1890.29  5617.8 1894.47
#Mann=3,-1,0
  4744.4    0.05       0  4989.4    0.03       0  5004.2    0.05       0
Bank Sta=4989.4,5004.2
Exp/Cntr=0.3,0.1

Type RM Length L Ch R = 1,78768,421,421,421
BEGIN DESCRIPTION:
Spring Creek 130.0
END DESCRIPTION:
XS GIS Cut Line= 3
      1659204.97      6880037.98      1659655.00      6880288.00
      1660254.98      6880288.00
#Sta/Elev= 30
  4484.9 1884.02  4610.8 1880.99  4661.1 1880.41  4770.9 1877.17  4816.7 1876.54
  4823.5 1875.76  4839.6 1875.52  4851.0 1874.57  4888.8 1873.12  4910.5 1871.54
  4919.6 1869.90  4932.2 1869.10  4964.3 1865.23  4970.0 1865.56  4976.8 1864.68
  4986.0 1864.99  5012.3 1862.81  5012.8 1862.31  5026.7 1862.31  5027.2 1862.81
  5029.7 1863.94  5049.7 1868.30  5129.7 1870.29  5159.7 1872.47  5259.7 1875.92
  5269.7 1875.45  5399.7 1879.62  5459.7 1882.96  5529.7 1889.06  5599.7 1893.22
#Mann=3,-1,0
  4484.9    0.05       0  5012.3    0.03       0  5027.2    0.05       0
Bank Sta=5012.3,5027.2
Exp/Cntr=0.3,0.1

Type RM Length L Ch R = 1,78347,190,190,190
BEGIN DESCRIPTION:
Spring Creek 129.0
END DESCRIPTION:
XS GIS Cut Line= 3
      1659212.64      6880473.59      1659657.08      6880709.70
      1660205.05      6880637.99
#Sta/Elev= 30
  4498.6 1878.00  4534.8 1877.71  4562.4 1876.71  4578.7 1876.80  4666.7 1874.27
  4672.3 1873.72  4726.9 1872.94  4814.9 1869.61  4886.5 1867.92  4897.1 1866.48
  4902.8 1867.31  4908.9 1865.59  4990.7 1863.21  4997.9 1860.89  5001.9 1860.89
  5002.3 1859.96  5002.8 1859.46  5016.8 1859.46  5017.3 1859.96  5019.9 1860.32
  5040.1 1868.43  5049.3 1869.81  5110.7 1869.80  5120.8 1869.24  5171.2 1869.64
  5262.0 1873.00  5359.8 1878.49  5413.3 1880.75  5473.8 1885.37  5554.5 1890.00
#Mann=3,-1,0
  4498.6    0.05       0  5002.3    0.03       0  5017.3    0.05       0
Bank Sta=5002.3,5017.3
Exp/Cntr=0.3,0.1

Type RM Length L Ch R = 1,78157,358,358,358
BEGIN DESCRIPTION:
Mapping XS fb312b8a
END DESCRIPTION:
XS GIS Cut Line= 2
      1659077.19      6880827.75      1660121.20      6880938.74
#Sta/Elev= 30
  4468.9 1877.18  4677.9 1869.92  4687.9 1870.03  4748.3 1868.23  4758.3 1867.38
  4778.4 1866.84  4802.9 1865.52  4808.6 1864.72  4828.7 1865.14  4848.8 1866.24
  4869.0 1866.04  4889.1 1866.53  4979.6 1863.86  4993.1 1862.87  5009.7 1859.19
  5022.4 1858.34  5022.9 1857.84  5036.9 1857.84  5037.4 1858.34  5050.0 1861.44
  5070.1 1867.33  5085.6 1867.65  5090.7 1866.84  5100.3 1866.19  5130.4 1866.39
  5251.1 1871.68  5275.8 1872.94  5311.4 1875.55  5361.7 1877.81  5518.8 1882.77
#Mann=3,-1,0
  4468.9    0.05       0  5022.4    0.03       0  5037.4    0.05       0
Bank Sta=5022.4,5037.4
Exp/Cntr=0.3,0.1

Type RM Length L Ch R = 1,77799,421,421,421
BEGIN DESCRIPTION:
Spring Creek 128.0
END DESCRIPTION:
XS GIS Cut Line= 3
      1659055.03      6881088.01      1659455.00      6881188.00
      1659927.88      6881234.00
#Sta/Elev= 30
  4587.6 1881.60  4605.6 1879.67  4652.0 1876.83  4688.1 1872.23  4693.2 1872.25
  4711.3 1870.38  4793.7 1865.31  4816.9 1864.30  4886.5 1863.51  4899.4 1862.87
  4907.1 1863.45  4927.7 1863.07  4935.5 1861.84  4969.0 1861.69  4981.8 1860.21
  4989.6 1861.51  5009.9 1861.07  5030.0 1861.33  5040.1 1859.47  5040.7 1858.90
  5041.2 1858.40  5055.5 1858.40  5056.0 1858.90  5060.2 1860.14  5090.3 1865.29
  5110.4 1866.03  5130.5 1867.90  5170.7 1869.60  5331.4 1873.88  5475.0 1876.37
#Mann=3,-1,0
  4587.6    0.05       0  5040.7    0.03       0  5056.0    0.05       0
Bank Sta=5040.7,5056
Exp/Cntr=0.3,0.1

Type RM Length L Ch R = 1,77378,206,206,206
BEGIN DESCRIPTION:
Spring Creek 127.0
END DESCRIPTION:
XS GIS Cut Line= 3
      1659004.95      6881437.99      1659205.00      6881488.00
      1660404.97      6881188.01
#Sta/Elev= 30
  4798.3 1879.24  4839.6 1876.02  4857.6 1872.88  4898.8 1868.24  4922.0 1866.94
  4945.2 1864.70  4953.0 1862.93  4978.8 1855.19  4979.3 1854.69  4993.7 1854.69
  4994.2 1855.19  5014.8 1856.29  5022.5 1857.72  5027.7 1856.48  5045.7 1860.63
  5063.8 1862.37  5110.2 1863.00  5146.2 1861.81  5210.7 1862.80  5275.1 1865.26
  5352.4 1869.16  5375.6 1869.37  5398.8 1870.62  5550.8 1871.83  5715.7 1874.50
  5764.7 1876.04  5769.9 1875.71  6094.6 1882.79  6189.9 1886.99  6241.4 1888.16
#Mann=3,-1,0
  4798.3    0.05       0  4978.8    0.05       0  4994.2    0.05       0
Bank Sta=4978.8,4994.2
Exp/Cntr=0.3,0.1

Type RM Length L Ch R = 1,77172,271,271,271
BEGIN DESCRIPTION:
Mapping XS 4a3d99d9
END DESCRIPTION:
XS GIS Cut Line= 3
      1658886.22      6881515.23      1659045.97      6881681.92
      1659806.38      6881654.15
#Sta/Elev= 30
  4658.8 1881.23  4716.6 1879.85  4759.0 1877.16  4815.4 1874.50  4836.7 1872.49
  4891.7 1870.33  4898.7 1869.38  4908.7 1869.37  4938.7 1866.46  4948.7 1864.63
  4978.8 1855.39  5001.1 1852.78  5001.6 1852.28  5016.0 1852.28  5016.5 1852.78
  5018.8 1854.55  5028.8 1857.65  5038.8 1860.03  5048.8 1860.79  5098.8 1860.86
  5148.9 1859.96  5188.9 1861.37  5198.9 1861.25  5228.9 1862.67  5248.9 1864.19
  5379.0 1866.43  5399.0 1867.04  5429.1 1868.85  5469.1 1870.16  5650.6 1870.75
#Mann=3,-1,0
  4658.8    0.05       0  5001.1    0.05       0  5016.5    0.05       0
Bank Sta=5001.1,5016.5
Exp/Cntr=0.3,0.1

Type RM Length L Ch R = 1,76901,454,454,454
BEGIN DESCRIPTION:
Spring Creek 126.0
END DESCRIPTION:
XS GIS Cut Line= 3
      1658905.05      6881838.02      1659205.00      6881938.00
      1659966.13      6881727.06
#Sta/Elev= 30
  4691.4 1877.05  4744.1 1872.38  4796.8 1869.59  4838.9 1865.29  4891.6 1862.68
  4923.3 1858.07  4933.8 1858.17  4944.3 1855.81  4954.9 1852.68  4957.7 1850.93
  4958.2 1850.43  4972.6 1850.43  4973.1 1850.93  4976.0 1852.43  5004.9 1854.61
  5018.0 1854.81  5024.7 1855.76  5038.7 1856.71  5090.6 1857.63  5111.3 1858.47
  5163.2 1858.52  5211.7 1861.51  5251.2 1863.14  5364.4 1864.57  5484.9 1867.96
  5557.6 1868.61  5625.2 1868.46  5630.4 1868.96  5659.5 1868.64  5797.4 1870.51
#Mann=3,-1,0
  4691.4    0.05       0  4957.7    0.03       0  4973.1    0.05       0
Bank Sta=4957.7,4973.1
Exp/Cntr=0.3,0.1

Type RM Length L Ch R = 1,76447,419,419,419
BEGIN DESCRIPTION:
Spring Creek 125.0
END DESCRIPTION:
XS GIS Cut Line= 3
      1658655.02      6881988.01      1659255.00      6882338.00
      1659705.02      6882588.01
#Sta/Elev= 30
  4305.6 1888.97  4319.2 1888.13  4334.9 1885.61  4430.9 1878.72  4502.4 1871.69
  4554.1 1867.98  4612.8 1865.54  4736.0 1861.88  4794.7 1858.87  4853.4 1857.36
  4884.4 1857.60  4919.2 1855.66  4965.1 1854.83  4992.3 1851.91  5003.1 1851.98
  5008.2 1851.05  5020.6 1850.48  5021.1 1849.98  5038.8 1849.98  5039.3 1850.48
  5057.4 1853.20  5080.3 1858.42  5089.4 1858.77  5138.6 1857.74  5192.4 1858.41
  5214.1 1859.57  5235.9 1862.18  5301.1 1865.41  5425.8 1869.85  5515.0 1872.03
#Mann=3,-1,0
  4305.6    0.05       0  5020.6    0.03       0  5039.3    0.05       0
Bank Sta=5020.6,5039.3
Exp/Cntr=0.3,0.1

Type RM Length L Ch R = 1,76028,438,438,438
BEGIN DESCRIPTION:
Spring Creek 124.0
END DESCRIPTION:
XS GIS Cut Line= 3
      1658405.01      6882288.01      1659005.00      6882638.00
      1659704.98      6882738.00
#Sta/Elev= 30
  4312.1 1906.70  4315.0 1906.70  4319.9 1904.60  4335.2 1901.86  4341.4 1899.93
  4378.7 1894.22  4464.7 1884.59  4480.4 1881.50  4532.1 1876.74  4576.3 1870.64
  4619.3 1865.80  4671.0 1862.73  4801.2 1859.23  4832.6 1857.51  4838.4 1856.78
  4859.9 1850.12  4867.8 1849.65  4897.1 1851.77  4934.4 1852.03  4955.9 1851.36
  4968.0 1847.93  4968.5 1847.43  4986.7 1847.93  5003.8 1853.37  5047.1 1855.46
  5138.0 1856.89  5218.8 1855.86  5259.2 1856.52  5471.4 1867.17  5713.8 1873.70
#Mann=3,-1,0
  4312.1    0.05       0  4968.0    0.03       0  4986.7    0.05       0
Bank Sta=4968,4986.7
Exp/Cntr=0.3,0.1

Type RM Length L Ch R = 1,75590,380,380,380
BEGIN DESCRIPTION:
Spring Creek 123.0
END DESCRIPTION:
XS GIS Cut Line= 3
      1658204.97      6882687.99      1658705.00      6882888.00
      1659405.04      6883088.01
#Sta/Elev= 30
  4456.4 1916.20  4471.2 1915.19  4525.1 1905.75  4564.1 1896.22  4603.2 1888.90
  4662.4 1881.79  4725.7 1871.15  4779.5 1863.69  4801.1 1858.61  4818.6 1855.78
  4848.2 1854.42  4962.6 1854.18  4973.4 1852.77  4980.1 1849.78  4982.9 1847.42
  4983.4 1846.92  5001.6 1847.42  5005.3 1848.15  5050.8 1848.02  5118.4 1852.00
  5171.7 1852.80  5203.0 1851.65  5223.8 1852.22  5255.0 1854.16  5275.8 1857.50
  5286.2 1858.15  5336.9 1859.48  5381.1 1861.84  5453.9 1863.82  5723.0 1868.34
#Mann=3,-1,0
  4456.4    0.05       0  4982.9    0.03       0  5001.6    0.05       0
Bank Sta=4982.9,5001.6
Exp/Cntr=0.3,0.1

Type RM Length L Ch R = 1,75210,168,168,168
BEGIN DESCRIPTION:
Spring Creek 122.0
END DESCRIPTION:
XS GIS Cut Line= 3
      1658174.46      6882990.96      1658598.06      6883237.48
      1659154.96      6883288.00
#Sta/Elev= 30
  4503.0 1895.60  4515.2 1892.53  4538.3 1888.81  4588.5 1883.72  4610.0 1880.99
  4625.7 1877.38  4641.5 1876.05  4684.5 1866.13  4706.0 1863.42  4727.5 1859.25
  4743.2 1853.94  4780.5 1848.28  4829.3 1847.19  4839.2 1847.69  4845.0 1849.24
  4850.8 1848.50  4860.7 1850.23  4866.5 1849.05  4882.2 1851.17  4946.8 1846.97
  4979.3 1843.11  4979.8 1842.61  4998.1 1843.11  5030.2 1844.12  5040.2 1845.90
  5054.8 1852.79  5060.3 1854.21  5090.5 1855.60  5170.8 1857.77  5552.3 1864.36
#Mann=3,-1,0
  4503.0    0.05       0  4979.3    0.03       0  4998.1    0.05       0
Bank Sta=4979.3,4998.1
Exp/Cntr=0.3,0.1

Type RM Length L Ch R = 1,75042,350,350,350
BEGIN DESCRIPTION:
Mapping XS 525cef45
END DESCRIPTION:
XS GIS Cut Line= 2
      1658101.56      6883195.83      1658951.09      6883556.44
#Sta/Elev= 30
  4545.3 1888.21  4581.6 1885.78  4640.9 1880.01  4646.8 1878.14  4670.0 1874.72
  4701.1 1867.91  4755.4 1859.98  4793.7 1851.15  4831.5 1849.96  4907.5 1850.02
  4922.9 1848.31  4940.1 1849.48  4983.6 1849.86  5005.3 1846.50  5016.2 1847.47
  5028.4 1845.77  5028.5 1844.73  5029.0 1844.23  5047.3 1844.73  5052.1 1847.52
  5059.6 1848.90  5070.3 1849.35  5081.4 1852.65  5099.4 1853.85  5113.9 1852.91
  5146.5 1853.10  5222.6 1854.41  5244.3 1855.17  5252.2 1856.35  5468.2 1859.03
#Mann=3,-1,0
  4545.3    0.05       0  5028.5    0.03       0  5047.3    0.05       0
Bank Sta=5028.5,5047.3
Exp/Cntr=0.3,0.1

Type RM Length L Ch R = 1,74692,451,451,451
BEGIN DESCRIPTION:
Spring Creek 121.0
END DESCRIPTION:
XS GIS Cut Line= 3
      1658105.01      6883538.01      1658305.00      6883638.00
      1659205.03      6884238.02
#Sta/Elev= 30
  4781.8 1869.69  4826.5 1863.53  4885.2 1858.19  4907.6 1854.51  4924.3 1848.06
  4938.3 1845.66  4997.0 1845.39  5002.6 1844.94  5003.5 1842.10  5004.0 1841.60
  5022.3 1842.10  5041.4 1845.47  5049.0 1845.40  5064.0 1847.65  5085.0 1848.67
  5221.7 1850.03  5250.3 1849.17  5265.3 1849.98  5271.3 1849.06  5280.3 1849.48
  5286.3 1848.43  5301.3 1849.43  5316.4 1848.82  5358.4 1851.19  5481.6 1853.47
  5502.7 1855.22  5595.8 1858.60  5942.8 1866.77  5978.9 1869.10  6087.1 1872.99
#Mann=3,-1,0
  4781.8    0.05       0  5003.5    0.03       0  5022.3    0.05       0
Bank Sta=5003.5,5022.3
Exp/Cntr=0.3,0.1

Type RM Length L Ch R = 1,74241,440,440,440
BEGIN DESCRIPTION:
Spring Creek 120.0
END DESCRIPTION:
XS GIS Cut Line= 3
      1657955.00      6883888.00      1658155.00      6884038.00
      1658901.78      6884333.98
#Sta/Elev= 30
  4754.9 1863.24  4776.8 1861.43  4833.0 1854.85  4883.0 1851.68  4912.2 1848.12
  4958.9 1840.73  4959.4 1840.23  4977.5 1840.23  4978.0 1840.73  4991.4 1840.83
  5001.8 1841.85  5019.8 1841.94  5058.7 1844.98  5068.4 1845.27  5103.5 1844.26
  5112.5 1845.40  5122.4 1845.82  5127.8 1845.39  5152.1 1847.02  5157.5 1846.83
  5198.5 1848.75  5211.6 1850.30  5241.6 1852.06  5381.4 1855.17  5392.1 1855.80
  5403.4 1855.60  5628.8 1860.49  5692.5 1862.46  5697.8 1862.18  5808.2 1865.01
#Mann=3,-1,0
  4754.9    0.05       0  4958.9    0.03       0  4978.0    0.05       0
Bank Sta=4958.9,4978
Exp/Cntr=0.3,0.1

Type RM Length L Ch R = 1,73801,474,474,474
BEGIN DESCRIPTION:
Spring Creek 119.0
END DESCRIPTION:
XS GIS Cut Line= 3
      1657804.99      6883937.96      1658005.00      6884438.00
      1658255.02      6884738.03
#Sta/Elev= 30
  4470.7 1866.97  4546.1 1861.63  4563.6 1859.59  4610.8 1857.10  4641.7 1854.22
  4664.6 1853.92  4686.1 1852.74  4707.7 1850.17  4730.6 1848.65  4793.8 1846.69
  4838.3 1846.58  4880.0 1845.52  4901.6 1843.98  4911.0 1842.87  4916.4 1841.39
  4923.1 1841.02  4964.8 1840.27  4999.8 1838.67  5012.5 1838.85  5013.3 1838.17
  5013.8 1837.67  5032.1 1837.67  5032.6 1838.17  5045.1 1839.01  5065.9 1845.51
  5073.7 1846.97  5129.7 1851.53  5250.7 1855.80  5265.0 1855.56  5399.8 1859.18
#Mann=3,-1,0
  4470.7    0.05       0  5013.3    0.05       0  5032.6    0.05       0
Bank Sta=5013.3,5032.6
Exp/Cntr=0.3,0.1

Type RM Length L Ch R = 1,73327,441,441,441
BEGIN DESCRIPTION:
Spring Creek 118.0
END DESCRIPTION:
XS GIS Cut Line= 3
      1657555.00      6884237.98      1657655.00      6884738.00
      1657905.01      6884988.01
#Sta/Elev= 30
  4484.9 1856.26  4525.7 1854.47  4546.1 1854.26  4597.1 1852.46  4699.1 1846.45
  4739.9 1845.79  4750.1 1844.92  4770.5 1844.30  4821.5 1843.97  4841.9 1844.25
  4852.1 1843.63  4882.6 1843.02  4913.2 1841.07  4923.4 1839.92  4964.2 1838.83
  4974.4 1837.20  4992.3 1836.02  5009.0 1835.56  5013.4 1834.75  5013.9 1834.25
  5032.3 1834.25  5032.8 1834.75  5037.3 1839.35  5051.4 1843.53  5093.8 1846.88
  5136.2 1849.32  5164.5 1850.54  5221.1 1852.27  5277.7 1854.52  5348.4 1856.41
#Mann=3,-1,0
  4484.9    0.05       0  5013.4    0.05       0  5032.8    0.05       0
Bank Sta=5013.4,5032.8
Exp/Cntr=0.3,0.1

Type RM Length L Ch R = 1,72886,418,418,418
BEGIN DESCRIPTION:
Spring Creek 117.0
END DESCRIPTION:
XS GIS Cut Line= 3
      1657164.03      6884414.58      1657305.00      6884988.00
      1657444.78      6885354.24
#Sta/Elev= 30
  4415.0 1851.85  4449.4 1851.83  4542.1 1850.25  4573.0 1848.70  4644.7 1847.04
  4686.2 1844.20  4717.2 1842.99  4821.1 1841.97  4933.4 1839.44  4940.6 1838.68
  4954.0 1834.53  4964.3 1832.80  4972.4 1832.50  4972.9 1832.00  4991.3 1832.00
  4991.8 1832.50  5026.9 1836.47  5045.3 1838.03  5050.6 1839.18  5069.7 1839.96
  5080.7 1841.74  5091.1 1842.31  5130.1 1843.38  5190.3 1846.65  5208.9 1846.83
  5239.7 1848.85  5245.1 1848.47  5283.8 1850.43  5390.8 1853.68  5397.5 1854.27
#Mann=3,-1,0
  4415.0    0.05       0  4972.4    0.03       0  4991.8    0.05       0
Bank Sta=4972.4,4991.8
Exp/Cntr=0.3,0.1

Type RM Length L Ch R = 1,72468,429,429,429
BEGIN DESCRIPTION:
Spring Creek 116.0
END DESCRIPTION:
XS GIS Cut Line= 3
      1656555.01      6884588.01      1656955.00      6885188.00
      1657154.97      6885387.97
#Sta/Elev= 30
  4283.3 1852.48  4305.8 1851.60  4383.9 1850.29  4492.1 1847.63  4607.8 1844.29
  4636.3 1842.13  4657.4 1838.22  4679.9 1836.81  4723.5 1836.76  4744.5 1838.12
  4780.6 1839.01  4824.1 1837.65  4852.7 1838.25  4888.7 1837.94  4909.8 1837.40
  4939.8 1835.25  4968.3 1834.29  4975.9 1833.65  4981.2 1832.02  4981.7 1831.52
  5000.1 1831.52  5000.6 1832.02  5007.9 1832.25  5032.7 1837.99  5061.0 1840.59
  5075.1 1841.01  5117.5 1845.02  5160.0 1846.48  5244.8 1851.04  5287.2 1852.32
#Mann=3,-1,0
  4283.3    0.05       0  4981.2    0.03       0  5000.6    0.05       0
Bank Sta=4981.2,5000.6
Exp/Cntr=0.3,0.1

Type RM Length L Ch R = 1,72039,480,480,480
BEGIN DESCRIPTION:
Spring Creek 115.0
END DESCRIPTION:
XS GIS Cut Line= 3
      1656455.00      6884738.00      1656555.00      6885288.00
      1656654.99      6885587.96
#Sta/Elev= 30
  4442.1 1849.09  4726.7 1843.18  4787.7 1840.65  4828.3 1837.90  4848.7 1837.18
  4869.0 1833.93  4879.1 1834.18  4899.5 1835.58  4916.0 1834.77  4940.1 1835.04
  4960.5 1834.63  4974.4 1832.91  4980.8 1830.14  4988.8 1828.91  4989.3 1828.41
  5007.8 1828.41  5008.3 1828.91  5011.7 1829.59  5022.2 1833.95  5032.7 1837.40
  5053.8 1838.79  5085.4 1839.71  5106.5 1839.75  5127.6 1840.80  5138.1 1840.64
  5201.4 1843.16  5233.0 1845.60  5243.6 1845.70  5264.6 1847.03  5317.3 1849.10
#Mann=3,-1,0
  4442.1    0.05       0  4988.8    0.03       0  5008.3    0.05       0
Bank Sta=4988.8,5008.3
Exp/Cntr=0.3,0.1

Type RM Length L Ch R = 1,71559,470,470,470
BEGIN DESCRIPTION:
Spring Creek 114.0
END DESCRIPTION:
XS GIS Cut Line= 3
      1655505.02      6884788.02      1656105.00      6885388.00
      1656304.99      6885737.99
#Sta/Elev= 30
  4151.5 1848.73  4236.3 1846.68  4363.6 1844.91  4391.9 1844.04  4434.3 1843.96
  4448.5 1843.38  4505.0 1842.46  4646.4 1841.04  4759.6 1838.98  4802.0 1837.64
  4886.9 1836.64  4915.1 1835.22  4943.4 1832.88  4957.6 1831.34  4976.0 1827.71
  4976.5 1827.21  4995.3 1827.21  4995.8 1827.71  4996.5 1828.41  5002.9 1828.41
  5007.9 1830.98  5023.0 1832.06  5103.7 1834.14  5153.3 1835.91  5161.2 1835.81
  5308.8 1843.33  5336.2 1845.38  5357.8 1847.81  5373.6 1848.45  5403.1 1850.41
#Mann=3,-1,0
  4151.5    0.05       0  4976.0    0.03       0  4995.8    0.05       0
Bank Sta=4976,4995.8
Exp/Cntr=0.3,0.1

Type RM Length L Ch R = 1,71089,160,160,160
BEGIN DESCRIPTION:
Spring Creek 113.0
END DESCRIPTION:
XS GIS Cut Line= 3
      1654952.26      6885209.72      1655705.00      6885588.00
      1656166.95      6885893.36
#Sta/Elev= 30
  4157.5 1844.68  4316.2 1840.36  4395.6 1836.72  4485.1 1835.26  4561.8 1836.81
  4628.8 1836.61  4768.3 1833.75  4790.6 1832.21  4807.4 1832.74  4813.0 1832.18
  4820.9 1833.06  4902.3 1829.60  4941.3 1829.70  4955.2 1830.65  4967.7 1829.13
  4968.2 1828.63  4987.5 1829.13  4991.6 1829.71  4997.2 1829.14  5022.5 1829.47
  5049.6 1831.40  5094.8 1831.35  5173.0 1834.60  5188.1 1834.64  5194.0 1835.62
  5224.2 1836.69  5230.2 1837.57  5404.7 1843.54  5467.9 1847.66  5553.7 1851.77
#Mann=3,-1,0
  4157.5    0.05       0  4967.7    0.03       0  4987.5    0.05       0
Bank Sta=4967.7,4987.5
Exp/Cntr=0.3,0.1

Type RM Length L Ch R = 1,70929,417,417,417
BEGIN DESCRIPTION:
Spring Creek 112.0
END DESCRIPTION:
XS GIS Cut Line= 3
      1654941.77      6885358.99      1655549.44      6885664.56
      1656007.32      6885973.28
#Sta/Elev= 30
  4278.7 1840.78  4416.1 1838.22  4505.4 1835.42  4555.6 1832.77  4617.0 1833.47
  4684.0 1833.12  4750.9 1831.55  4773.3 1830.78  4778.9 1829.97  4823.5 1828.73
  4868.2 1829.63  4890.5 1829.22  4912.8 1830.01  4972.8 1830.19  5013.8 1827.80
  5014.3 1827.30  5033.2 1827.30  5033.7 1827.80  5037.9 1829.89  5044.7 1830.38
  5050.8 1832.01  5074.1 1834.43  5116.7 1835.08  5173.7 1837.06  5218.6 1837.45
  5303.3 1839.94  5311.6 1839.52  5332.6 1841.01  5440.5 1844.18  5511.1 1848.22
#Mann=3,-1,0
  4278.7    0.05       0  5013.8    0.03       0  5033.7    0.05       0
Bank Sta=5013.8,5033.7
Exp/Cntr=0.3,0.1

Type RM Length L Ch R = 1,70512,355,355,355
BEGIN DESCRIPTION:
Mapping XS 42e02b95
END DESCRIPTION:
XS GIS Cut Line= 3
      1654868.91      6885449.30      1655032.08      6885563.87
      1655497.38      6886279.17
#Sta/Elev= 30
  4469.0 1840.29  4580.1 1834.54  4594.9 1835.05  4601.0 1834.67  4630.6 1834.78
  4687.0 1833.72  4768.7 1831.16  4810.9 1829.02  4826.0 1828.68  4847.1 1827.27
  4868.2 1827.47  4889.3 1826.35  4904.5 1826.84  4911.9 1826.04  4925.6 1826.14
  4940.7 1827.38  4947.7 1827.19  4951.8 1825.74  4952.3 1825.24  4971.3 1825.24
  4971.8 1825.74  4976.9 1826.96  4992.1 1826.40  5019.3 1826.78  5034.3 1827.86
  5055.4 1830.18  5091.6 1831.77  5106.7 1831.81  5143.0 1832.96  5521.7 1837.14
#Mann=3,-1,0
  4469.0    0.05       0  4951.8    0.03       0  4971.8    0.05       0
Bank Sta=4951.8,4971.8
Exp/Cntr=0.3,0.1

Type RM Length L Ch R = 1,70157,556,556,556
BEGIN DESCRIPTION:
Spring Creek 111.0
END DESCRIPTION:
XS GIS Cut Line= 3
      1654660.55      6885376.35      1654905.00      6885988.00
      1655664.00      6886622.87
#Sta/Elev= 30
  4335.6 1846.86  4488.1 1842.76  4757.4 1833.39  4823.3 1829.77  4832.8 1828.85
  4854.3 1824.96  4865.1 1824.23  4867.1 1823.10  4867.6 1822.60  4886.6 1822.60
  4887.1 1823.10  4908.1 1824.51  4940.4 1824.57  4949.8 1823.74  4955.2 1824.49
  4979.5 1824.87  4984.9 1823.91  4991.6 1823.69  5015.8 1824.08  5030.1 1826.02
  5036.6 1827.81  5050.9 1829.59  5129.0 1830.82  5143.3 1831.51  5264.3 1832.81
  5371.0 1833.06  5377.5 1833.68  5619.5 1836.69  5895.4 1840.74  5983.8 1842.53
#Mann=3,-1,0
  4335.6    0.05       0  4867.1    0.05       0  4887.1    0.05       0
Bank Sta=4867.1,4887.1
Exp/Cntr=0.3,0.1

Type RM Length L Ch R = 1,69601,529,529,529
BEGIN DESCRIPTION:
Spring Creek 110.0
END DESCRIPTION:
XS GIS Cut Line= 3
      1654055.02      6886088.01      1654455.00      6886288.00
      1655528.63      6886855.54
#Sta/Elev= 30
  4545.8 1871.99  4568.1 1868.34  4604.5 1865.61  4649.2 1860.66  4688.3 1854.06
  4783.4 1843.30  4805.7 1838.39  4822.5 1832.81  4836.5 1829.42  4889.6 1819.11
  4911.9 1821.03  4925.9 1824.04  4948.3 1823.06  4956.7 1821.57  4962.2 1819.19
  4969.0 1818.24  4969.5 1817.74  4989.1 1818.24  5001.2 1819.62  5023.2 1819.54
  5038.2 1822.94  5050.8 1827.70  5067.2 1828.26  5230.5 1828.88  5413.7 1830.83
  5430.1 1830.04  5435.7 1830.83  5474.1 1831.64  5858.9 1837.02  6207.4 1840.13
#Mann=3,-1,0
  4545.8    0.05       0  4969.0    0.03       0  4989.1    0.05       0
Bank Sta=4969,4989.1
Exp/Cntr=0.3,0.1

Type RM Length L Ch R = 1,69072,535,535,535
BEGIN DESCRIPTION:
Spring Creek 109.0
END DESCRIPTION:
XS GIS Cut Line= 3
      1653914.03      6886487.48      1654155.00      6886688.00
      1655420.49      6886917.95
#Sta/Elev= 30
  4685.7 1844.16  4708.2 1843.83  4729.0 1842.26  4778.5 1839.98  4786.3 1840.05
  4792.8 1838.76  4815.0 1836.94  4835.8 1834.47  4878.8 1831.82  4934.7 1823.81
  4956.9 1819.68  4963.4 1819.52  4971.2 1817.90  4975.5 1814.46  4976.0 1813.96
  4995.1 1813.96  4995.6 1814.46  5031.0 1816.03  5060.2 1820.98  5079.3 1822.34
  5182.1 1825.02  5395.6 1827.94  5414.8 1827.19  5426.1 1828.09  5478.3 1828.86
  5531.7 1828.84  5638.4 1830.24  5643.5 1829.89  5913.9 1834.32  6285.4 1838.88
#Mann=3,-1,0
  4685.7    0.05       0  4975.5    0.05       0  4995.6    0.05       0
Bank Sta=4975.5,4995.6
Exp/Cntr=0.3,0.1

Type RM Length L Ch R = 1,68537,500,500,500
BEGIN DESCRIPTION:
Spring Creek 108.0
END DESCRIPTION:
XS GIS Cut Line= 3
      1653105.03      6886388.03      1653905.00      6887138.00
      1655455.02      6888688.02
#Sta/Elev= 30
  3897.1 1875.65  4052.6 1864.07  4088.3 1859.47  4215.3 1853.66  4293.4 1845.93
  4512.7 1832.19  4689.6 1827.12  4901.6 1823.01  4929.9 1821.55  4944.1 1817.96
  4948.1 1814.80  4948.6 1814.30  4968.3 1814.80  5007.8 1818.89  5064.3 1814.86
  5106.8 1820.53  5120.9 1820.65  5149.2 1817.06  5163.3 1817.17  5205.8 1820.10
  5234.1 1819.78  5262.3 1822.34  5884.6 1827.66  6153.3 1831.95  6464.4 1841.31
  6605.8 1848.31  6846.3 1865.00  7001.8 1881.42  7143.2 1892.69  7185.7 1893.64
#Mann=3,-1,0
  3897.1    0.05       0  4948.1    0.03       0  4968.3    0.05       0
Bank Sta=4948.1,4968.3
Exp/Cntr=0.3,0.1

Type RM Length L Ch R = 1,68037,578,578,578
BEGIN DESCRIPTION:
Spring Creek 107.0
END DESCRIPTION:
XS GIS Cut Line= 3
      1653304.99      6886787.98      1653705.00      6887588.00
      1655254.99      6888987.99
#Sta/Elev= 30
  4111.7 1851.97  4164.8 1846.33  4209.5 1839.07  4335.3 1827.18  4447.1 1824.12
  4872.0 1818.89  4908.3 1815.32  4953.0 1814.95  4969.8 1813.02  4973.4 1811.16
  4973.9 1810.66  4994.2 1811.16  5009.5 1812.12  5027.4 1817.91  5048.4 1819.13
  5091.0 1819.76  5303.2 1816.93  5395.8 1820.23  5451.9 1820.20  5544.6 1823.42
  5919.7 1829.87  6380.0 1842.89  6507.1 1849.49  6627.4 1859.10  6719.3 1864.37
  6804.5 1871.63  6875.5 1879.85  6910.6 1881.82  6932.3 1884.48  7094.8 1894.28
#Mann=3,-1,0
  4111.7    0.05       0  4973.4    0.03       0  4994.2    0.05       0
Bank Sta=4973.4,4994.2
Exp/Cntr=0.3,0.1

Type RM Length L Ch R = 1,67459,543,543,543
BEGIN DESCRIPTION:
Spring Creek 106.0
END DESCRIPTION:
XS GIS Cut Line= 3
      1652604.97      6887187.97      1653355.00      6887988.00
      1654155.00      6888788.00
#Sta/Elev= 30
  3923.8 1866.52  3973.4 1860.94  4022.8 1851.26  4058.4 1846.21  4072.6 1843.56
  4100.9 1836.44  4107.7 1833.84  4121.9 1831.61  4157.1 1827.28  4192.7 1824.31
  4298.7 1821.20  4581.8 1818.28  4744.7 1814.75  4815.0 1815.72  4829.2 1817.07
  4871.7 1815.85  4907.3 1812.46  4942.5 1812.31  4949.8 1810.94  4992.3 1811.47
  4999.2 1810.98  5002.9 1809.25  5003.4 1808.75  5023.7 1809.25  5034.6 1812.11
  5062.9 1816.43  5232.6 1814.01  5374.0 1818.79  5713.4 1824.47  6151.8 1838.17
#Mann=3,-1,0
  3923.8    0.05       0  5002.9    0.05       0  5023.7    0.05       0
Bank Sta=5002.9,5023.7
Exp/Cntr=0.3,0.1

Type RM Length L Ch R = 1,66916,512,512,512
BEGIN DESCRIPTION:
Spring Creek 105.0
END DESCRIPTION:
XS GIS Cut Line= 3
      1652497.38      6887706.24      1652856.58      6887991.67
      1654455.02      6889538.02
#Sta/Elev= 30
  4541.2 1861.21  4569.1 1857.90  4583.5 1849.46  4589.9 1849.16  4598.0 1845.09
  4604.3 1844.54  4626.8 1836.95  4633.2 1836.53  4647.6 1830.31  4697.3 1823.17
  4711.7 1819.53  4811.0 1813.58  4903.9 1814.43  4953.6 1813.14  4978.3 1806.32
  4978.8 1805.82  4999.3 1806.32  5067.1 1808.86  5074.1 1811.69  5081.3 1810.48
  5088.2 1813.81  5116.5 1814.55  5215.6 1813.43  5816.7 1819.34  6417.7 1834.91
  6756.5 1847.79  6842.1 1853.80  7004.7 1860.83  7174.5 1873.06  7224.0 1874.79
#Mann=3,-1,0
  4541.2    0.05       0  4978.3    0.05       0  4999.3    0.05       0
Bank Sta=4978.3,4999.3
Exp/Cntr=0.3,0.1

Type RM Length L Ch R = 1,66404,529,529,529
BEGIN DESCRIPTION:
Spring Creek 104.0
END DESCRIPTION:
XS GIS Cut Line= 3
      1652405.01      6887938.03      1652505.00      6888338.00
      1654054.97      6889737.97
#Sta/Elev= 30
  4588.2 1861.80  4652.6 1858.18  4693.8 1851.74  4729.9 1843.91  4763.4 1839.37
  4771.1 1837.39  4784.0 1832.09  4858.7 1811.43  4876.8 1810.30  4918.0 1812.27
  4928.3 1810.39  4941.2 1805.85  4959.1 1805.39  4959.6 1804.89  4980.1 1805.39
  5014.3 1806.90  5036.0 1811.74  5071.1 1812.87  5198.9 1814.01  5354.3 1813.54
  5368.5 1814.48  5538.9 1814.52  5743.7 1816.43  5949.2 1819.94  6218.2 1826.75
  6586.6 1841.29  6735.3 1850.19  6884.0 1856.90  7053.6 1869.38  7089.1 1870.18
#Mann=3,-1,0
  4588.2    0.05       0  4959.1    0.03       0  4980.1    0.05       0
Bank Sta=4959.1,4980.1
Exp/Cntr=0.3,0.1

Type RM Length L Ch R = 1,65875,588,588,588
BEGIN DESCRIPTION:
Spring Creek 103.0
END DESCRIPTION:
XS GIS Cut Line= 3
      1652105.00      6888138.01      1652055.00      6888538.00
      1653304.98      6890087.97
#Sta/Elev= 30
  4595.9 1840.82  4666.4 1839.31  4726.9 1836.32  4757.1 1832.25  4794.9 1824.53
  4888.1 1815.38  4918.4 1810.78  4948.6 1804.81  4956.2 1806.00  4958.3 1804.64
  4958.8 1804.14  4979.3 1804.64  4988.9 1807.85  5027.0 1808.85  5055.8 1807.01
  5070.2 1809.53  5084.6 1810.46  5468.4 1810.80  5924.0 1813.89  6023.4 1815.51
  6399.3 1825.29  6463.5 1827.95  6485.6 1830.04  6549.6 1832.99  6677.5 1842.79
  6776.7 1847.76  6840.7 1853.59  6890.3 1856.64  6954.3 1863.35  6990.2 1865.09
#Mann=3,-1,0
  4595.9    0.05       0  4958.3    0.03       0  4979.3    0.05       0
Bank Sta=4958.3,4979.3
Exp/Cntr=0.3,0.1

Type RM Length L Ch R = 1,65287,386,386,386
BEGIN DESCRIPTION:
Spring Creek 102.0
END DESCRIPTION:
XS GIS Cut Line= 3
      1651005.00      6888138.00      1651605.00      6888888.00
      1653154.98      6890287.98
#Sta/Elev= 30
  4039.5 1856.50  4096.3 1853.15  4167.6 1846.62  4259.6 1835.53  4346.1 1830.00
  4423.7 1821.69  4487.7 1816.93  4538.1 1814.98  4914.3 1809.39  4935.9 1808.13
  4964.0 1800.50  4975.9 1799.71  4976.4 1799.21  4996.9 1799.71  5000.0 1803.02
  5007.1 1804.40  5049.7 1808.30  5290.3 1807.20  5304.5 1806.94  5325.4 1803.97
  5347.1 1806.54  5375.5 1807.08  5948.7 1812.31  6409.0 1825.74  6543.5 1832.86
  6649.6 1841.92  6763.2 1847.26  6890.2 1859.00  6989.6 1866.06  7088.6 1870.57
#Mann=3,-1,0
  4039.5    0.05       0  4975.9    0.03       0  4996.9    0.05       0
Bank Sta=4975.9,4996.9
Exp/Cntr=0.3,0.1

Type RM Length L Ch R = 1,64901,789,789,789
BEGIN DESCRIPTION:
Spring Creek 101.0
END DESCRIPTION:
XS GIS Cut Line= 3
      1650959.16      6888407.61      1651375.83      6889174.98
      1652555.00      6890388.00
#Sta/Elev= 30
  4133.1 1831.79  4240.6 1826.56  4278.7 1822.49  4372.5 1816.44  4475.4 1812.60
  4633.2 1808.65  4867.9 1806.35  4955.3 1807.14  4971.5 1803.75  4977.2 1800.51
  4982.9 1798.80  4983.4 1798.30  5003.9 1798.80  5005.2 1799.68  5029.0 1801.24
  5043.2 1805.61  5050.3 1806.72  5248.2 1804.68  5736.1 1809.12  5891.8 1811.88
  6111.1 1818.02  6139.4 1819.11  6252.4 1826.79  6379.7 1837.13  6492.9 1843.20
  6507.0 1845.24  6563.6 1848.90  6613.2 1853.97  6662.6 1856.83  6698.0 1857.62
#Mann=3,-1,0
  4133.1    0.05       0  4982.9    0.03       0  5003.9    0.05       0
Bank Sta=4982.9,5003.9
Exp/Cntr=0.3,0.1

Type RM Length L Ch R = 1,64112,429,429,429
BEGIN DESCRIPTION:
Spring Creek 100.0
END DESCRIPTION:
XS GIS Cut Line= 3
      1650824.44      6888703.35      1651256.85      6889681.76
      1652154.96      6890337.97
#Sta/Elev= 30
  3930.3 1828.69  4017.8 1824.44  4023.3 1822.88  4064.4 1819.63  4087.7 1816.71
  4099.4 1813.97  4154.0 1807.53  4230.6 1804.37  4389.2 1803.34  4799.1 1805.64
  4830.5 1804.37  4842.8 1800.02  4859.3 1798.48  4864.8 1800.16  4905.9 1802.12
  4911.4 1803.51  4952.2 1803.63  4963.4 1801.55  4970.7 1797.71  4971.2 1797.21
  4991.9 1797.71  4995.2 1799.53  5047.0 1801.32  5067.9 1803.63  5159.8 1803.27
  5239.3 1806.69  5790.3 1816.21  5904.2 1822.28  6040.2 1833.49  6112.3 1836.57
#Mann=3,-1,0
  3930.3    0.05       0  4970.7    0.03       0  4991.9    0.05       0
Bank Sta=4970.7,4991.9
Exp/Cntr=0.3,0.1

Type RM Length L Ch R = 1,63683,723,723,723
BEGIN DESCRIPTION:
Spring Creek 99.0
END DESCRIPTION:
XS GIS Cut Line= 3
      1650555.00      6888787.99      1650955.00      6889938.00
      1651104.99      6890737.97
#Sta/Elev= 30
  3786.7 1847.20  3926.7 1835.58  3988.9 1827.09  4062.0 1821.08  4114.9 1806.80
  4164.9 1798.74  4232.4 1800.67  4305.5 1799.51  4351.5 1801.16  4408.4 1800.43
  4657.2 1802.70  4887.8 1800.90  4931.8 1802.52  4951.3 1801.05  4962.9 1797.35
  4972.5 1796.68  4973.0 1796.18  4993.7 1796.68  5024.6 1798.40  5045.0 1804.22
  5075.5 1806.77  5095.9 1805.72  5135.7 1807.79  5251.0 1808.55  5289.2 1806.17
  5380.7 1809.52  5563.9 1825.29  5655.4 1830.37  5706.3 1835.80  5818.2 1842.04
#Mann=3,-1,0
  3786.7    0.05       0  4972.5    0.03       0  4993.7    0.05       0
Bank Sta=4972.5,4993.7
Exp/Cntr=0.3,0.1

Type RM Length L Ch R = 1,62960,459,459,459
BEGIN DESCRIPTION:
Mapping XS 27f436e4
END DESCRIPTION:
XS GIS Cut Line= 2
      1650572.71      6888955.14      1650520.71      6890064.62
#Sta/Elev= 30
  4379.5 1834.02  4402.4 1832.58  4437.4 1827.01  4442.4 1827.73  4522.5 1820.19
  4542.5 1816.69  4602.6 1802.38  4622.6 1798.73  4632.6 1797.95  4654.3 1797.02
  4682.7 1798.27  4712.7 1797.80  4772.8 1799.24  4792.8 1798.63  4842.9 1799.67
  4912.9 1796.44  4923.0 1796.21  4943.0 1797.22  4952.4 1793.48  4952.9 1792.98
  4973.7 1793.48  5013.1 1795.87  5053.1 1795.95  5078.1 1797.83  5133.2 1798.01
  5193.3 1802.15  5373.5 1803.22  5393.5 1804.39  5413.5 1803.33  5490.2 1803.61
#Mann=3,-1,0
  4379.5    0.05       0  4952.4    0.03       0  4973.7    0.05       0
Bank Sta=4952.4,4973.7
Exp/Cntr=0.3,0.1

Type RM Length L Ch R = 1,62501,472,472,472
BEGIN DESCRIPTION:
Mapping XS e8474281
END DESCRIPTION:
XS GIS Cut Line= 3
      1650212.64      6889056.96      1650278.61      6889480.53
      1650740.20      6890740.36
#Sta/Elev= 30
  4766.3 1831.16  4787.6 1829.54  4813.5 1825.77  4881.4 1822.70  4919.2 1819.29
  4929.3 1817.07  4944.3 1810.82  4949.5 1805.28  4969.8 1796.96  4979.9 1791.14
  4989.4 1788.42  4989.9 1787.92  5010.8 1788.42  5012.2 1793.56  5020.4 1796.04
  5060.8 1797.98  5131.7 1797.52  5370.7 1800.46  5447.9 1800.21  5523.3 1801.63
  5807.0 1804.12  5979.5 1801.93  6045.8 1804.74  6204.0 1806.47  6304.4 1809.52
  6385.1 1813.84  6395.9 1815.24  6415.8 1815.66  6446.3 1818.37  6536.7 1823.69
#Mann=3,-1,0
  4766.3    0.05       0  4989.4    0.05       0  5010.8    0.05       0
Bank Sta=4989.4,5010.8
Exp/Cntr=0.3,0.1

Type RM Length L Ch R = 1,62029,520,520,520
BEGIN DESCRIPTION:
Spring Creek 98.0
END DESCRIPTION:
XS GIS Cut Line= 3
      1649719.58      6889202.74      1649855.00      6889488.00
      1650169.14      6890050.33
#Sta/Elev= 30
  4684.6 1818.47  4759.0 1818.40  4827.1 1814.90  4849.9 1811.78  4872.6 1807.11
  4878.6 1804.43  4895.3 1801.18  4911.8 1799.44  4918.1 1797.80  4934.0 1795.97
  4940.8 1794.61  4946.3 1792.19  4958.3 1789.17  4958.8 1788.67  4979.2 1788.67
  4979.7 1789.17  4986.2 1789.45  4997.6 1793.12  5003.2 1793.12  5014.1 1795.09
  5023.3 1795.26  5067.8 1794.45  5073.5 1795.02  5103.5 1795.23  5148.9 1793.68
  5176.3 1795.57  5192.3 1795.04  5300.8 1797.41  5500.7 1800.43  5644.5 1801.45
#Mann=3,-1,0
  4684.6    0.05       0  4958.3    0.03       0  4979.7    0.05       0
Bank Sta=4958.3,4979.7
Exp/Cntr=0.3,0.1

Type RM Length L Ch R = 1,61509,403,403,403
BEGIN DESCRIPTION:
Spring Creek 97.0
END DESCRIPTION:
XS GIS Cut Line= 3
      1649654.99      6889288.04      1649555.00      6889738.00
      1649580.00      6889962.98
#Sta/Elev= 30
  4532.8 1816.24  4584.0 1814.96  4614.7 1812.60  4644.2 1809.58  4649.3 1809.41
  4665.9 1806.37  4692.8 1800.39  4697.9 1800.85  4706.9 1799.16  4736.4 1796.58
  4741.5 1796.52  4747.9 1795.69  4778.6 1794.76  4833.7 1794.34  4840.1 1793.91
  4891.3 1793.22  4920.8 1792.56  4925.9 1792.07  4942.5 1792.46  4963.0 1792.34
  4996.3 1790.71  5013.2 1789.41  5013.7 1788.91  5034.2 1788.91  5034.7 1789.41
  5044.0 1792.02  5064.2 1796.35  5154.7 1796.77  5174.8 1797.82  5220.1 1797.46
#Mann=3,-1,0
  4532.8    0.05       0  5013.2    0.03       0  5034.7    0.05       0
Bank Sta=5013.2,5034.7
Exp/Cntr=0.3,0.1

Type RM Length L Ch R = 1,61106,326,326,326
BEGIN DESCRIPTION:
Spring Creek 96.0
END DESCRIPTION:
XS GIS Cut Line= 3
      1648955.02      6889238.05      1649146.67      6889716.65
      1649270.86      6890095.15
#Sta/Elev= 30
  4461.9 1823.81  4500.9 1820.30  4515.7 1820.08  4525.1 1818.47  4554.7 1815.54
  4601.9 1813.82  4692.0 1808.17  4709.6 1805.55  4716.2 1802.72  4740.4 1796.78
  4745.8 1796.35  4752.7 1794.42  4770.0 1792.78  4794.3 1791.94  4871.2 1792.21
  4901.9 1790.58  4925.0 1791.98  4946.6 1790.66  4961.1 1792.16  4968.1 1792.04
  4975.5 1789.93  4980.8 1789.93  4986.1 1788.40  5007.2 1787.26  5007.7 1786.76
  5028.7 1787.26  5063.1 1789.13  5081.6 1793.77  5105.2 1794.87  5375.8 1795.37
#Mann=3,-1,0
  4461.9    0.05       0  5007.2    0.03       0  5028.7    0.05       0
Bank Sta=5007.2,5028.7
Exp/Cntr=0.3,0.1

Type RM Length L Ch R = 1,60780,524,524,524
BEGIN DESCRIPTION:
Mapping XS f25e8c7a
END DESCRIPTION:
XS GIS Cut Line= 3
      1648757.78      6889230.53      1648778.61      6889536.09
      1648980.02      6890013.04
#Sta/Elev= 30
  4528.2 1815.26  4535.7 1814.53  4560.8 1813.67  4565.8 1813.90  4595.8 1812.78
  4656.0 1812.02  4704.5 1810.45  4726.1 1810.60  4756.2 1809.69  4766.2 1809.82
  4806.3 1808.25  4826.4 1808.20  4858.3 1806.77  4869.1 1805.40  4880.0 1803.34
  4887.4 1799.57  4911.1 1792.84  4923.4 1791.13  4945.7 1790.70  4976.9 1785.62
  4977.4 1785.12  4998.0 1785.12  4998.5 1785.62  5022.2 1786.75  5064.2 1790.69
  5122.5 1792.82  5175.3 1793.53  5199.1 1793.31  5216.5 1793.95  5352.2 1793.97
#Mann=3,-1,0
  4528.2    0.05       0  4976.9    0.03       0  4998.5    0.05       0
Bank Sta=4976.9,4998.5
Exp/Cntr=0.3,0.1

Type RM Length L Ch R = 1,60256,362,362,362
BEGIN DESCRIPTION:
Spring Creek 95.0
END DESCRIPTION:
XS GIS Cut Line= 3
      1648323.77      6889459.73      1648577.22      6889869.42
      1649132.79      6891230.55
#Sta/Elev= 30
  4497.8 1809.11  4584.8 1807.00  4658.1 1803.10  4752.7 1793.34  4779.8 1789.12
  4837.7 1786.41  4883.8 1786.25  4919.1 1789.12  4979.6 1789.77  4985.2 1788.35
  4990.6 1790.56  5009.2 1784.27  5014.6 1787.66  5021.2 1782.37  5021.7 1781.87
  5042.8 1782.37  5062.7 1787.81  5068.1 1786.27  5086.0 1791.76  5092.1 1792.08
  5291.2 1790.09  5330.0 1791.49  5538.4 1790.33  5645.4 1791.72  5669.3 1791.59
  5690.9 1789.10  5712.5 1791.25  6079.7 1798.44  6228.1 1808.25  6449.7 1813.64
#Mann=3,-1,0
  4497.8    0.05       0  5021.2    0.03       0  5042.8    0.05       0
Bank Sta=5021.2,5042.8
Exp/Cntr=0.3,0.1

Type RM Length L Ch R = 1,59894,565,565,565
BEGIN DESCRIPTION:
Spring Creek 94.0
END DESCRIPTION:
XS GIS Cut Line= 3
      1648054.98      6889537.97      1648255.00      6889888.00
      1648816.46      6891163.77
#Sta/Elev= 30
  4596.7 1823.59  4663.7 1817.13  4722.7 1809.71  4830.7 1801.91  4852.3 1798.64
  4868.1 1792.77  4911.3 1785.23  4932.9 1787.85  4976.8 1788.01  4991.9 1785.63
  4997.0 1782.57  5002.6 1782.57  5003.4 1780.40  5003.9 1779.90  5025.1 1780.40
  5032.1 1785.16  5043.6 1787.66  5084.3 1790.10  5165.2 1790.95  5578.3 1789.63
  5589.8 1788.50  5659.3 1789.41  5729.3 1788.51  5856.9 1790.47  5895.7 1789.16
  5972.2 1789.25  6060.0 1794.60  6281.0 1804.28  6327.7 1808.57  6393.7 1812.08
#Mann=3,-1,0
  4596.7    0.05       0  5003.4    0.05       0  5025.1    0.05       0
#XS Ineff=2,0
       0                 5241.10    0.00 1801.09
Permanent Ineff=
       F       F
Bank Sta=5003.4,5025.1
Exp/Cntr=0.3,0.1

Type RM Length L Ch R = 1,59329,292,292,292
BEGIN DESCRIPTION:
Spring Creek 93.0
END DESCRIPTION:
XS GIS Cut Line= 3
      1647542.51      6889647.22      1647705.00      6889938.00
      1648556.38      6891112.47
#Sta/Elev= 30
  4666.8 1824.89  4705.2 1822.19  4736.4 1818.49  4742.9 1816.60  4786.3 1812.65
  4845.7 1805.14  4910.8 1800.42  4942.6 1793.94  4948.5 1791.02  4954.2 1791.68
  4977.0 1787.14  4986.2 1779.62  4986.7 1779.12  5007.9 1779.62  5028.1 1783.02
  5063.7 1784.78  5086.4 1783.83  5185.2 1786.68  5407.5 1788.51  5938.6 1788.22
  6001.6 1785.66  6016.3 1787.11  6102.1 1786.72  6173.3 1791.69  6273.7 1795.50
  6282.3 1794.53  6296.8 1795.26  6317.8 1798.57  6382.8 1804.56  6450.5 1807.40
#Mann=3,-1,0
  4666.8    0.05       0  4986.2    0.05       0  5007.9    0.05       0
#XS Ineff=2,0
       0                 5281.90    0.00 1797.55
Permanent Ineff=
       F       F
Bank Sta=4986.2,5007.9
Exp/Cntr=0.3,0.1
