--- Threemile Creek.prj (project) ---

Proj Title=Threemile Creek Base Level Engineering
Current Plan=p01
Default Exp/Contr=0.3,0.1
English Units
Geom File=g01
Flow File=f01
Plan File=p01
BEGIN DESCRIPTION:
Threemile Creek
END DESCRIPTION:

--- Threemile Creek.p01 (plan) ---

Plan Title=Multiple Run
Short Identifier=Multiple
Geom File=g01
Flow File=f01
Subcritical Flow
K Sum by GR= 0
Std Step Tol= 0.01
Critical Tol= 0.01
Num of Std Step Trials= 20
Max Error Tol= 0.3
Flow Tol Ratio= 0.001
Split Flow NTrial= 30
Split Flow Tol= 0.02
Split Flow Ratio= 0.02
Log Output Level= 0
Friction Slope Method= 1
Unsteady Friction Slope Method= 2
Unsteady Bridges Friction Slope Method= 1
Parabolic Critical Depth
Global Vel Dist=  1 , 1 , 1
Global Log Level= 0
CheckData=True
Encroach Param= -1, 0, 0, 0
BEGIN DESCRIPTION:
Multiple Run
END DESCRIPTION:

--- Threemile Creek.f01 (steady flow) ---

Flow Title=Multiple
Number of Profiles=7
Profile Names=10-year,25-year,50-year,1pct_min,100-year,1pct_plu,500-year
River Rch & RM= Threemile Creek,Reach-1,40786
     206     281     342     208     414     827     614
River Rch & RM= Threemile Creek,Reach-1,40523
     256     353     433     264     528    1053     793
River Rch & RM= Threemile Creek,Reach-1,36228
     508     727     914     570    1138    2271    1790
River Rch & RM= Threemile Creek,Reach-1,32198
     594     855    1078     675    1348    2689    2133
River Rch & RM= Threemile Creek,Reach-1,27616
     667     963    1217     763    1523    3038    2418
River Rch & RM= Threemile Creek,Reach-1,20214
     698    1010    1278     802    1601    3195    2548
River Rch & RM= Threemile Creek,Reach-1,16566
    1010    1486    1902    1207    2408    4805    3914
River Rch & RM= Threemile Creek,Reach-1,12035
    1081    1595    2046    1301    2596    5180    4238
River Rch & RM= Threemile Creek,Reach-1,8058
    1155    1709    2196    1399    2791    5569    4570
River Rch & RM= Threemile Creek,Reach-1,3543
    1163    1720    2210    1407    2808    5603    4596
Boundary for River Rch & Prof#=Threemile Creek,Reach-1,1
Up Type=0
Dn Type=3
Dn Slope=0.003
Boundary for River Rch & Prof#=Threemile Creek,Reach-1,2
Up Type=0
Dn Type=3
Dn Slope=0.003
Boundary for River Rch & Prof#=Threemile Creek,Reach-1,3
Up Type=0
Dn Type=3
Dn Slope=0.003
Boundary for River Rch & Prof#=Threemile Creek,Reach-1,4
Up Type=0
Dn Type=3
Dn Slope=0.003
Boundary for River Rch & Prof#=Threemile Creek,Reach-1,5
Up Type=0
Dn Type=3
Dn Slope=0.003
Boundary for River Rch & Prof#=Threemile Creek,Reach-1,6
Up Type=0
Dn Type=3
Dn Slope=0.003
Boundary for River Rch & Prof#=Threemile Creek,Reach-1,7
Up Type=0
Dn Type=3
Dn Slope=0.003

--- Threemile Creek.g01 (geometry) ---

Geom Title=Existing Conditions

River Reach=Threemile Creek,Reach-1
Reach XY= 30
      1650305.00      6934588.00      1649834.97      6934237.39
      1648916.87      6934636.27      1647957.43      6933743.52
      1647210.89      6933786.04      1646723.20      6933388.12
      1646127.86      6933614.43      1645214.70      6934977.26
      1643602.70      6935293.83      1643049.32      6936086.03
      1642189.84      6935437.52      1641160.86      6936085.94
      1640265.55      6935339.10      1639064.79      6936577.48
      1638258.46      6936846.47      1638901.25      6937836.45
      1637218.62      6938824.78      1637082.14      6939961.53
      1636329.92      6940288.20      1635156.46      6939891.54
      1634199.10      6941735.77      1632013.44      6941691.41
      1631361.06      6942429.86      1629252.56      6943343.52
      1628653.37      6944034.06      1626980.08      6944338.20
      1626160.47      6944040.44      1625425.66      6942007.43
      1623961.03      6941939.62      1623255.00      6943688.00

Type RM Length L Ch R = 1,40786,263,263,263
BEGIN DESCRIPTION:
Threemile Creek 78.0
END DESCRIPTION:
XS GIS Cut Line= 3
      1650680.01      6934112.99      1650305.00      6934588.00
      1650155.00      6934887.99
#Sta/Elev= 30
  4394.8 1757.74  4479.8 1756.48  4487.8 1756.71  4593.6 1754.64  4608.0 1754.78
  4694.2 1752.43  4744.3 1751.70  4779.6 1750.44  4814.8 1750.06  4893.4 1746.85
  4922.3 1747.56  4949.5 1746.84  4986.4 1746.94  4996.8 1746.01  5002.8 1746.01
  5012.0 1744.92  5012.2 1744.42  5015.7 1744.42  5016.0 1744.92  5022.4 1745.29
  5030.7 1746.95  5044.7 1748.38  5075.5 1749.67  5081.1 1750.31  5148.1 1751.38
  5170.5 1752.54  5178.9 1752.33  5282.3 1754.38  5299.1 1755.19  5335.4 1755.24
#Mann=3,-1,0
  4394.8    0.05       0  5012.0    0.03       0  5016.0    0.05       0
Bank Sta=5012,5016
Exp/Cntr=0.3,0.1

Type RM Length L Ch R = 1,40523,316,316,316
BEGIN DESCRIPTION:
Mapping XS 0e097248
END DESCRIPTION:
XS GIS Cut Line= 2
      1650363.13      6934137.11      1649896.97      6934686.62
#Sta/Elev= 30
  4567.8 1754.72  4595.2 1754.31  4602.7 1754.66  4609.2 1754.09  4652.1 1753.48
  4715.8 1751.42  4752.1 1749.83  4758.6 1750.09  4815.8 1748.04  4850.9 1747.65
  4865.2 1747.10  4879.5 1747.07  4886.0 1746.66  4914.6 1746.26  4943.2 1744.10
  4949.7 1744.40  4957.5 1745.26  4964.0 1745.07  4978.3 1743.91  4990.6 1743.50
  4990.8 1743.00  4994.3 1743.00  4994.6 1743.50  5006.9 1744.30  5027.9 1746.95
  5056.3 1748.66  5084.9 1748.78  5127.7 1749.60  5205.7 1750.37  5288.4 1750.49
#Mann=3,-1,0
  4567.8    0.05       0  4990.6    0.03       0  4994.6    0.05       0
Bank Sta=4990.6,4994.6
Exp/Cntr=0.3,0.1

Type RM Length L Ch R = 1,40207,446,446,446
BEGIN DESCRIPTION:
Threemile Creek 77.0
END DESCRIPTION:
XS GIS Cut Line= 3
      1649905.00      6934088.05      1649905.00      6934238.00
      1649826.68      6934678.74
#Sta/Elev= 30
  4844.9 1753.59  4847.4 1753.59  4854.9 1752.46  4864.9 1751.49  4924.9 1749.48
  4964.9 1747.21  4984.9 1744.67  4990.4 1742.51  4990.6 1742.01  4994.1 1742.01
  4994.4 1742.51  5021.8 1743.76  5055.8 1744.58  5075.8 1744.37  5086.3 1743.56
  5106.6 1743.44  5139.9 1744.81  5147.2 1745.44  5157.4 1745.78  5167.5 1745.69
  5177.7 1746.19  5228.5 1746.62  5247.9 1747.36  5253.0 1747.09  5299.6 1748.28
  5312.0 1748.09  5360.5 1749.13  5391.0 1749.17  5411.3 1749.64  5442.5 1749.60
#Mann=3,-1,0
  4844.9    0.05       0  4990.4    0.03       0  4994.4    0.05       0
Bank Sta=4990.4,4994.4
Exp/Cntr=0.3,0.1

Type RM Length L Ch R = 1,39761,419,419,419
BEGIN DESCRIPTION:
Threemile Creek 76.0
END DESCRIPTION:
XS GIS Cut Line= 3
      1649455.00      6934087.97      1649505.00      6934388.00
      1649706.05      6934804.67
#Sta/Elev= 30
  4701.3 1751.75  4721.6 1751.41  4741.9 1750.09  4782.4 1749.18  4802.7 1748.00
  4812.8 1748.13  4863.5 1747.03  4873.7 1746.29  4904.1 1745.34  4934.5 1743.13
  4964.9 1739.68  4970.5 1739.49  4970.8 1738.99  4974.3 1738.99  4974.5 1739.49
  4995.3 1741.12  5014.0 1741.91  5027.7 1741.79  5072.1 1742.74  5081.8 1743.31
  5087.4 1742.99  5094.3 1743.36  5132.6 1743.35  5160.9 1744.57  5206.0 1744.58
  5260.8 1745.71  5290.8 1745.61  5371.9 1747.18  5416.3 1747.25  5468.1 1748.87
#Mann=3,-1,0
  4701.3    0.05       0  4970.5    0.03       0  4974.5    0.05       0
Bank Sta=4970.5,4974.5
Exp/Cntr=0.3,0.1

Type RM Length L Ch R = 1,39342,409,409,409
BEGIN DESCRIPTION:
Threemile Creek 75.0
END DESCRIPTION:
XS GIS Cut Line= 3
      1649199.07      6934079.81      1649155.00      6934588.00
      1649390.88      6935018.29
#Sta/Elev= 30
  4489.7 1750.92  4648.5 1747.07  4748.9 1744.17  4779.0 1743.94  4809.1 1742.59
  4869.3 1742.01  4879.4 1741.20  4938.2 1739.78  4943.3 1740.05  4959.7 1739.60
  4969.7 1740.15  5007.9 1739.49  5020.6 1737.95  5020.9 1737.45  5024.4 1737.45
  5024.6 1737.95  5035.4 1739.89  5073.3 1740.16  5089.4 1740.88  5116.9 1741.32
  5138.7 1742.50  5160.5 1742.85  5198.4 1744.54  5258.1 1745.00  5279.9 1745.55
  5285.6 1746.08  5330.5 1746.12  5367.1 1747.16  5456.0 1748.59  5490.5 1749.97
#Mann=3,-1,0
  4489.7    0.05       0  5020.6    0.03       0  5024.6    0.05       0
Bank Sta=5020.6,5024.6
Exp/Cntr=0.3,0.1

Type RM Length L Ch R = 1,38933,449,449,449
BEGIN DESCRIPTION:
Threemile Creek 74.0
END DESCRIPTION:
XS GIS Cut Line= 3
      1649354.97      6933738.04      1648855.00      6934538.00
      1648705.02      6934887.96
#Sta/Elev= 30
  4056.0 1762.57  4121.4 1759.95  4127.3 1760.08  4163.9 1757.72  4185.7 1756.93
  4331.3 1753.02  4352.5 1753.00  4563.0 1746.76  4608.4 1746.00  4614.3 1745.34
  4708.7 1743.25  4729.9 1742.30  4760.6 1741.98  4854.9 1739.69  4860.8 1739.10
  4905.0 1737.82  4949.2 1737.14  4970.5 1735.98  4983.7 1734.62  4984.0 1734.12
  4987.6 1734.12  4987.8 1734.62  5008.4 1735.99  5021.1 1737.75  5032.0 1738.37
  5042.9 1740.21  5075.5 1741.59  5119.0 1742.44  5236.9 1747.09  5380.1 1750.80
#Mann=3,-1,0
  4056.0    0.05       0  4983.7    0.03       0  4987.8    0.05       0
Bank Sta=4983.7,4987.8
Exp/Cntr=0.3,0.1

Type RM Length L Ch R = 1,38484,427,427,427
BEGIN DESCRIPTION:
Threemile Creek 73.0
END DESCRIPTION:
XS GIS Cut Line= 3
      1648955.00      6933938.00      1648605.00      6934188.00
      1648405.01      6934687.97
#Sta/Elev= 30
  4569.8 1748.96  4598.1 1747.99  4619.0 1747.87  4627.6 1747.30  4633.7 1747.48
  4734.5 1744.48  4749.2 1744.42  4791.0 1742.61  4841.4 1741.51  4906.5 1738.02
  4969.6 1732.64  4969.9 1732.14  4973.5 1732.14  4973.7 1732.64  4996.8 1733.75
  5039.0 1734.35  5053.8 1735.57  5075.3 1736.54  5139.9 1738.65  5146.7 1739.24
  5170.9 1739.57  5236.9 1742.19  5269.2 1742.63  5301.5 1744.06  5337.8 1744.39
  5398.4 1746.71  5409.2 1746.72  5445.5 1748.05  5475.2 1748.14  5538.4 1750.22
#Mann=3,-1,0
  4569.8    0.05       0  4969.6    0.03       0  4973.7    0.05       0
Bank Sta=4969.6,4973.7
Exp/Cntr=0.3,0.1

Type RM Length L Ch R = 1,38057,166,166,166
BEGIN DESCRIPTION:
Threemile Creek 72.0
END DESCRIPTION:
XS GIS Cut Line= 3
      1648805.03      6933737.98      1648255.00      6933988.00
      1648255.00      6934538.01
#Sta/Elev= 30
  4395.2 1749.12  4409.5 1748.22  4478.7 1746.27  4530.3 1745.20  4538.0 1744.66
  4553.4 1744.63  4599.6 1743.11  4622.6 1742.87  4628.1 1742.13  4645.7 1741.93
  4658.9 1741.19  4713.8 1739.77  4735.8 1738.59  4869.8 1733.58  4887.3 1733.28
  4944.5 1733.61  5017.3 1731.25  5017.6 1730.75  5021.2 1730.75  5021.5 1731.25
  5049.4 1732.44  5059.4 1733.26  5069.4 1735.25  5079.4 1735.94  5139.4 1737.00
  5199.4 1740.10  5219.4 1740.44  5259.4 1742.05  5449.4 1745.28  5549.4 1747.64
#Mann=3,-1,0
  4395.2    0.05       0  5017.3    0.03       0  5021.5    0.05       0
Bank Sta=5017.3,5021.5
Exp/Cntr=0.3,0.1

Type RM Length L Ch R = 1,37891,280,280,280
BEGIN DESCRIPTION:
Mapping XS a59297ea
END DESCRIPTION:
XS GIS Cut Line= 2
      1648331.88      6933603.26      1647975.19      6934103.15
#Sta/Elev= 30
  4650.0 1740.63  4687.1 1739.75  4693.2 1739.14  4701.9 1739.36  4708.0 1738.80
  4722.7 1738.46  4729.5 1737.83  4773.1 1735.63  4859.2 1732.77  4915.7 1731.98
  4945.2 1732.36  5022.3 1730.47  5022.6 1729.97  5026.2 1729.97  5026.5 1730.47
  5046.0 1731.09  5052.2 1731.92  5073.5 1733.72  5102.5 1734.75  5117.3 1736.35
  5123.4 1736.26  5152.9 1737.42  5182.4 1737.81  5188.6 1737.51  5203.3 1737.84
  5209.5 1737.58  5218.1 1738.13  5224.2 1737.71  5232.8 1738.05  5264.1 1738.05
#Mann=3,-1,0
  4650.0    0.05       0  5022.3    0.05       0  5026.5    0.05       0
Bank Sta=5022.3,5026.5
Exp/Cntr=0.3,0.1

Type RM Length L Ch R = 1,37611,370,370,370
BEGIN DESCRIPTION:
Threemile Creek 71.0
END DESCRIPTION:
XS GIS Cut Line= 3
      1648167.80      6933447.03      1647905.00      6933738.00
      1647915.21      6934217.81
#Sta/Elev= 30
  4608.9 1737.10  4632.9 1737.29  4639.7 1736.89  4675.5 1737.10  4682.3 1736.73
  4703.9 1736.84  4710.7 1736.31  4739.1 1736.05  4745.8 1735.35  4767.4 1734.58
  4880.3 1732.38  4944.6 1731.64  4979.7 1730.79  4997.6 1729.85  5028.9 1729.17
  5029.2 1728.67  5032.8 1728.67  5033.1 1729.17  5071.0 1729.91  5131.0 1730.51
  5191.0 1732.42  5231.0 1734.52  5271.0 1735.70  5351.1 1736.53  5391.1 1737.56
  5401.1 1737.43  5431.1 1738.41  5441.1 1738.24  5461.1 1739.39  5480.9 1739.47
#Mann=3,-1,0
  4608.9    0.05       0  5028.9    0.05       0  5033.1    0.05       0
Bank Sta=5028.9,5033.1
Exp/Cntr=0.3,0.1

Type RM Length L Ch R = 1,37241,89,89,89
BEGIN DESCRIPTION:
Mapping XS e2c2c362
END DESCRIPTION:
XS GIS Cut Line= 2
      1647595.34      6933450.04      1647521.73      6934114.68
#Sta/Elev= 30
  4721.2 1741.09  4739.3 1740.59  4749.3 1744.52  4759.4 1746.04  4772.1 1745.21
  4799.6 1742.25  4809.7 1740.65  4839.9 1733.38  4849.9 1732.26  4857.7 1731.68
  4862.8 1731.90  4870.1 1731.07  4900.2 1724.69  4910.3 1723.58  4920.4 1723.22
  5079.1 1722.81  5079.4 1722.31  5083.2 1722.31  5083.5 1722.81  5129.8 1722.86
  5141.7 1723.21  5161.8 1724.80  5182.0 1727.19  5262.4 1733.63  5311.2 1735.30
  5316.3 1735.21  5342.9 1736.31  5353.0 1737.09  5383.2 1737.36  5389.9 1737.69
#Mann=3,-1,0
  4721.2    0.05       0  5079.1    0.03       0  5083.5    0.05       0
Bank Sta=5079.1,5083.5
Exp/Cntr=0.3,0.1

Type RM Length L Ch R = 1,37152,70,70,70
BEGIN DESCRIPTION:
Threemile Creek 70.0
END DESCRIPTION:
XS GIS Cut Line= 3
      1647512.87      6933411.00      1647478.15      6933734.34
      1647437.09      6934084.44
#Sta/Elev= 30
  4670.5 1739.68  4700.0 1738.79  4717.8 1739.73  4768.1 1739.25  4792.1 1738.29
  4828.4 1738.84  4878.7 1737.82  4884.2 1737.03  4889.2 1738.25  4939.0 1738.10
  4959.2 1737.68  4976.3 1735.73  4981.3 1738.22  5039.7 1738.03  5065.2 1734.83
  5070.3 1737.41  5110.1 1737.21  5148.4 1735.75  5153.5 1737.34  5200.8 1737.76
  5231.0 1736.14  5236.7 1734.04  5241.7 1735.69  5248.9 1733.32  5249.2 1732.82
  5253.0 1732.82  5253.3 1733.32  5261.2 1734.08  5281.3 1734.04  5348.2 1736.98
#Mann=3,-1,0
  4670.5    0.05       0  5248.9    0.03       0  5253.3    0.05       0
Bank Sta=5248.9,5253.3
Exp/Cntr=0.3,0.1

Type RM Length L Ch R = 1,37082,255,255,255
BEGIN DESCRIPTION:
Mapping XS 00dbed5e
END DESCRIPTION:
XS GIS Cut Line= 2
      1647436.91      6933404.52      1647378.32      6934088.11
#Sta/Elev= 30
  4664.3 1737.22  4728.0 1735.69  4738.1 1735.39  4744.1 1734.87  4758.1 1735.01
  4808.3 1732.04  4838.4 1731.30  4857.9 1730.27  4868.5 1729.18  4938.8 1727.12
  4968.9 1725.53  4976.7 1724.70  4986.8 1724.43  4987.1 1723.93  4990.9 1723.93
  4991.2 1724.43  5029.1 1725.84  5049.2 1727.10  5069.3 1727.74  5079.3 1728.59
  5129.5 1729.85  5189.7 1731.90  5209.2 1732.88  5219.8 1734.38  5229.9 1735.41
  5239.9 1733.42  5249.9 1733.35  5270.0 1733.88  5310.1 1735.94  5350.4 1736.81
#Mann=3,-1,0
  4664.3    0.05       0  4986.8    0.03       0  4991.2    0.05       0
Bank Sta=4986.8,4991.2
Exp/Cntr=0.3,0.1

Type RM Length L Ch R = 1,36827,174,174,174
BEGIN DESCRIPTION:
Mapping XS 21bfb3a6
END DESCRIPTION:
XS GIS Cut Line= 2
      1647356.64      6933421.81      1647052.82      6933996.89
#Sta/Elev= 30
  4616.3 1732.91  4635.4 1731.41  4645.9 1731.54  4679.9 1730.80  4695.8 1729.92
  4712.1 1729.48  4717.8 1728.85  4734.1 1728.71  4739.8 1729.19  4770.3 1728.26
  4866.2 1726.83  4894.7 1726.01  4917.4 1726.23  4940.0 1725.44  4962.6 1725.12
  4998.3 1723.85  5018.1 1723.64  5018.4 1723.14  5022.2 1723.14  5022.6 1723.64
  5036.7 1724.08  5042.3 1723.83  5058.7 1724.04  5064.4 1726.15  5075.1 1727.28
  5087.0 1729.38  5119.1 1731.18  5168.8 1733.37  5185.1 1734.57  5266.7 1736.22
#Mann=3,-1,0
  4616.3    0.05       0  5018.1    0.03       0  5022.6    0.05       0
Bank Sta=5018.1,5022.6
Exp/Cntr=0.3,0.1

Type RM Length L Ch R = 1,36653,109,109,109
BEGIN DESCRIPTION:
Threemile Creek 69.0
END DESCRIPTION:
XS GIS Cut Line= 3
      1647293.69      6933315.49      1647055.00      6933638.00
      1646931.27      6933907.96
#Sta/Elev= 30
  4598.5 1732.39  4691.8 1729.74  4700.2 1729.86  4777.4 1727.86  4785.8 1728.08
  4792.0 1727.63  4821.3 1727.34  4856.8 1726.21  4963.2 1724.88  4992.4 1722.36
  5002.5 1722.19  5008.5 1722.70  5014.0 1722.68  5021.7 1721.91  5029.2 1721.73
  5029.6 1721.23  5033.4 1721.23  5033.7 1721.73  5043.7 1722.20  5060.0 1722.13
  5076.7 1724.26  5088.5 1726.71  5098.7 1727.66  5111.5 1727.94  5142.7 1730.26
  5164.7 1731.39  5203.5 1732.60  5209.0 1733.88  5249.5 1734.78  5296.7 1735.25
#Mann=3,-1,0
  4598.5    0.05       0  5029.2    0.03       0  5033.7    0.05       0
Bank Sta=5029.2,5033.7
Exp/Cntr=0.3,0.1

Type RM Length L Ch R = 1,36544,160,160,160
BEGIN DESCRIPTION:
Mapping XS c12786ef
END DESCRIPTION:
XS GIS Cut Line= 3
      1647213.42      6933351.58      1646994.70      6933523.42
      1646852.21      6933844.69
#Sta/Elev= 30
  4680.6 1730.08  4704.7 1729.26  4719.2 1729.29  4748.1 1728.48  4762.5 1728.43
  4768.9 1727.99  4777.0 1728.06  4841.2 1725.80  4862.0 1725.64  4890.9 1724.59
  4897.2 1724.83  4905.3 1724.35  4969.8 1724.09  4998.5 1722.72  5016.3 1722.51
  5029.4 1721.30  5049.0 1720.78  5049.3 1720.28  5053.2 1720.28  5053.5 1720.78
  5062.2 1721.34  5073.8 1723.62  5106.0 1726.61  5143.6 1728.42  5149.7 1729.34
  5218.9 1732.19  5226.3 1732.74  5242.2 1732.77  5265.5 1733.94  5310.2 1734.50
#Mann=3,-1,0
  4680.6    0.05       0  5049.0    0.03       0  5053.5    0.05       0
Bank Sta=5049,5053.5
Exp/Cntr=0.3,0.1

Type RM Length L Ch R = 1,36384,156,156,156
BEGIN DESCRIPTION:
Mapping XS 552b0bde
END DESCRIPTION:
XS GIS Cut Line= 3
      1647174.29      6933350.24      1646896.55      6933426.18
      1646777.77      6933784.68
#Sta/Elev= 30
  4707.3 1729.03  4748.0 1728.43  4759.6 1727.78  4768.8 1727.88  4828.7 1725.50
  4851.7 1725.00  4908.0 1722.24  4913.9 1721.63  4942.5 1720.75  4947.7 1720.90
  4980.0 1719.42  4980.3 1718.92  4984.2 1718.92  4984.5 1719.42  5007.7 1719.95
  5028.8 1720.82  5077.9 1720.96  5083.2 1721.29  5102.5 1721.59  5134.1 1722.99
  5141.3 1723.75  5146.6 1723.21  5165.7 1723.93  5228.9 1728.30  5236.4 1728.63
  5241.7 1728.50  5250.0 1729.04  5292.1 1730.58  5313.2 1731.92  5372.9 1733.11
#Mann=3,-1,0
  4707.3    0.05       0  4980.0    0.03       0  4984.5    0.05       0
Bank Sta=4980,4984.5
Exp/Cntr=0.3,0.1

Type RM Length L Ch R = 1,36228,322,322,322
BEGIN DESCRIPTION:
Threemile Creek 68.0
END DESCRIPTION:
XS GIS Cut Line= 3
      1646655.00      6933188.01      1646755.00      6933388.00
      1646755.00      6933688.00
#Sta/Elev= 30
  4776.4 1727.95  4821.1 1726.54  4857.5 1724.58  4874.2 1722.90  4896.6 1722.13
  4910.6 1722.63  4924.5 1725.15  4932.9 1725.70  4941.3 1724.22  4946.9 1724.15
  4963.7 1720.20  4969.3 1719.64  4986.0 1712.98  5006.8 1712.66  5007.3 1712.16
  5012.8 1712.16  5013.3 1712.66  5020.0 1712.83  5040.0 1719.13  5070.0 1724.67
  5080.0 1723.33  5090.0 1722.91  5130.0 1723.28  5150.0 1722.61  5160.0 1723.73
  5190.0 1724.59  5220.0 1727.15  5250.0 1727.28  5290.0 1729.88  5300.0 1729.92
#Mann=3,-1,0
  4776.4    0.05       0  5006.8    0.05       0  5013.3    0.05       0
Bank Sta=5006.8,5013.3
Exp/Cntr=0.3,0.1

Type RM Length L Ch R = 1,35906,192,192,192
BEGIN DESCRIPTION:
Threemile Creek 67.0
END DESCRIPTION:
XS GIS Cut Line= 3
      1646503.75      6933020.41      1646442.99      6933426.18
      1646655.01      6933838.01
#Sta/Elev= 30
  4576.9 1734.00  4695.8 1729.80  4734.2 1727.34  4796.9 1726.17  4837.4 1724.79
  4877.8 1721.31  4918.3 1720.59  4948.6 1718.80  4958.7 1718.58  4968.8 1719.25
  4991.0 1719.52  5011.7 1719.30  5026.5 1718.49  5048.7 1719.22  5070.8 1718.36
  5076.0 1717.38  5076.5 1716.88  5082.0 1716.88  5082.5 1717.38  5093.0 1718.55
  5101.7 1720.39  5115.2 1721.13  5214.2 1721.82  5281.3 1725.25  5292.9 1726.64
  5315.4 1727.99  5347.8 1729.41  5397.8 1730.38  5419.9 1732.10  5450.4 1732.59
#Mann=3,-1,0
  4576.9    0.05       0  5076.0    0.03       0  5082.5    0.05       0
Bank Sta=5076,5082.5
Exp/Cntr=0.3,0.1

Type RM Length L Ch R = 1,35714,394,394,394
BEGIN DESCRIPTION:
Mapping XS f879980a
END DESCRIPTION:
XS GIS Cut Line= 2
      1646132.49      6933264.47      1646509.06      6933874.26
#Sta/Elev= 30
  4712.9 1724.94  4717.9 1724.94  4752.3 1723.19  4798.4 1721.95  4862.2 1721.48
  4869.8 1721.76  4883.5 1721.30  4950.9 1720.80  4963.9 1719.65  4972.2 1716.99
  4978.1 1715.93  4983.9 1715.42  4984.4 1714.92  4990.3 1714.92  4990.8 1715.42
  5008.8 1716.35  5036.0 1718.78  5066.8 1719.06  5116.7 1720.49  5146.0 1720.68
  5182.6 1720.16  5234.2 1720.16  5261.8 1720.69  5277.2 1721.22  5298.5 1723.33
  5313.9 1724.40  5363.5 1725.82  5408.5 1727.79  5414.4 1728.30  5429.6 1728.36
#Mann=3,-1,0
  4712.9    0.05       0  4983.9    0.03       0  4990.8    0.05       0
Bank Sta=4983.9,4990.8
Exp/Cntr=0.3,0.1

Type RM Length L Ch R = 1,35320,437,437,437
BEGIN DESCRIPTION:
Threemile Creek 66.0
END DESCRIPTION:
XS GIS Cut Line= 3
      1645805.01      6933538.01      1646055.00      6933788.00
      1646404.99      6934087.99
#Sta/Elev= 30
  4640.2 1733.86  4654.3 1733.59  4696.7 1729.63  4710.9 1728.67  4739.2 1728.37
  4767.5 1727.12  4781.6 1726.01  4795.7 1724.34  4838.2 1718.69  4880.6 1715.66
  4937.2 1717.26  4965.5 1716.84  4979.6 1716.07  4990.2 1714.87  5004.0 1714.73
  5004.5 1714.23  5010.5 1714.23  5011.0 1714.73  5021.7 1716.77  5036.0 1717.75
  5064.5 1719.08  5113.9 1720.52  5142.5 1721.98  5191.8 1723.10  5199.5 1723.64
  5220.4 1723.62  5256.6 1724.67  5263.2 1724.43  5334.5 1725.93  5454.7 1729.89
#Mann=3,-1,0
  4640.2    0.05       0  5004.0    0.03       0  5011.0    0.05       0
Bank Sta=5004,5011
Exp/Cntr=0.3,0.1

Type RM Length L Ch R = 1,34883,423,423,423
BEGIN DESCRIPTION:
Threemile Creek 65.0
END DESCRIPTION:
XS GIS Cut Line= 3
      1645705.01      6933838.04      1645755.00      6934088.00
      1646154.98      6934287.99
#Sta/Elev= 30
  4745.0 1727.17  4816.3 1725.36  4826.5 1724.09  4846.9 1722.25  4867.3 1720.89
  4877.5 1718.95  4918.3 1716.68  4928.5 1715.48  4969.3 1712.81  4979.5 1711.66
  4993.8 1711.11  4994.3 1710.61  5000.4 1710.61  5000.9 1711.11  5053.0 1715.06
  5075.4 1716.33  5097.7 1715.85  5134.1 1716.02  5215.1 1718.71  5223.5 1719.27
  5231.9 1719.04  5237.5 1719.67  5245.9 1719.69  5313.0 1721.86  5321.3 1722.17
  5326.9 1722.74  5357.7 1723.32  5388.4 1724.62  5416.4 1725.09  5447.1 1726.19
#Mann=3,-1,0
  4745.0    0.05       0  4993.8    0.03       0  5000.9    0.05       0
Bank Sta=4993.8,5000.9
Exp/Cntr=0.3,0.1

Type RM Length L Ch R = 1,34460,448,448,448
BEGIN DESCRIPTION:
Threemile Creek 64.0
END DESCRIPTION:
XS GIS Cut Line= 3
      1645355.02      6934288.02      1645555.00      6934438.00
      1645904.96      6934737.97
#Sta/Elev= 30
  4755.0 1726.52  4791.4 1725.58  4841.4 1722.33  4855.0 1721.01  4868.5 1718.91
  4918.5 1712.87  4933.1 1712.25  4968.5 1713.80  4976.8 1711.50  4987.8 1709.58
  4988.3 1709.08  4994.5 1709.08  4995.0 1709.58  4997.7 1709.75  5001.8 1711.22
  5008.3 1711.22  5012.1 1712.05  5054.9 1712.11  5083.4 1711.14  5097.2 1712.27
  5153.7 1715.40  5182.2 1717.64  5338.1 1721.56  5387.5 1723.55  5395.2 1724.24
  5401.7 1724.13  5430.3 1725.31  5438.0 1726.35  5452.2 1726.14  5465.9 1726.84
#Mann=3,-1,0
  4755.0    0.05       0  4987.8    0.03       0  4995.0    0.05       0
Bank Sta=4987.8,4995
Exp/Cntr=0.3,0.1

Type RM Length L Ch R = 1,34012,428,428,428
BEGIN DESCRIPTION:
Threemile Creek 63.0
END DESCRIPTION:
XS GIS Cut Line= 3
      1645155.03      6934588.03      1645355.00      6934788.00
      1645754.99      6934838.00
#Sta/Elev= 30
  4717.2 1724.14  4759.6 1722.41  4773.7 1720.88  4787.9 1719.91  4830.3 1714.75
  4872.7 1711.12  4901.0 1709.97  4943.4 1711.16  4971.7 1710.84  4985.9 1711.08
  4996.5 1709.05  5002.5 1709.05  5026.6 1708.00  5027.1 1707.50  5033.3 1707.50
  5033.8 1708.00  5037.8 1708.07  5050.4 1709.99  5070.5 1711.56  5090.7 1712.56
  5118.4 1715.23  5204.1 1716.80  5231.8 1716.75  5251.9 1717.72  5262.0 1717.70
  5284.7 1718.35  5302.3 1719.44  5342.6 1721.20  5372.9 1723.39  5403.1 1724.61
#Mann=3,-1,0
  4717.2    0.05       0  5026.6    0.03       0  5033.8    0.05       0
Bank Sta=5026.6,5033.8
Exp/Cntr=0.3,0.1

Type RM Length L Ch R = 1,33584,440,440,440
BEGIN DESCRIPTION:
Threemile Creek 62.0
END DESCRIPTION:
XS GIS Cut Line= 3
      1645005.01      6934688.05      1645055.00      6934988.00
      1645205.01      6935588.04
#Sta/Elev= 30
  4689.2 1724.11  4699.3 1723.68  4739.8 1720.34  4782.9 1718.11  4838.7 1713.69
  4904.6 1710.39  4932.5 1708.09  4942.6 1707.73  4965.4 1708.01  4973.0 1707.27
  4999.3 1707.25  4999.8 1706.75  5007.4 1706.75  5007.9 1707.25  5011.3 1707.63
  5034.5 1708.10  5044.8 1709.41  5057.7 1710.01  5065.4 1709.93  5075.8 1709.19
  5093.8 1709.11  5098.9 1709.52  5117.0 1709.17  5135.0 1710.11  5140.2 1709.87
  5176.3 1712.28  5395.3 1717.83  5457.1 1719.09  5477.8 1720.13  5611.8 1724.11
#Mann=3,-1,0
  4689.2    0.05       0  4999.3    0.03       0  5007.9    0.05       0
Bank Sta=4999.3,5007.9
Exp/Cntr=0.3,0.1

Type RM Length L Ch R = 1,33144,481,481,481
BEGIN DESCRIPTION:
Threemile Creek 61.0
END DESCRIPTION:
XS GIS Cut Line= 3
      1644755.01      6934787.96      1644655.00      6935088.00
      1644705.00      6935588.04
#Sta/Elev= 30
  4684.1 1720.27  4715.8 1719.11  4757.9 1716.44  4768.5 1716.20  4800.1 1714.09
  4810.6 1713.82  4831.7 1712.32  4937.1 1710.12  4958.2 1708.94  4968.7 1706.80
  5006.1 1705.10  5006.6 1704.60  5014.2 1704.60  5014.7 1705.10  5020.5 1706.53
  5030.5 1707.65  5053.1 1707.50  5060.7 1706.50  5070.7 1706.44  5110.9 1708.67
  5161.2 1710.21  5211.4 1710.60  5254.1 1710.29  5271.7 1710.99  5311.9 1711.58
  5349.6 1713.90  5354.6 1713.82  5372.2 1715.53  5392.3 1716.81  5502.9 1721.23
#Mann=3,-1,0
  4684.1    0.05       0  5006.1    0.05       0  5014.7    0.05       0
Bank Sta=5006.1,5014.7
Exp/Cntr=0.3,0.1

Type RM Length L Ch R = 1,32663,465,465,465
BEGIN DESCRIPTION:
Threemile Creek 60.0
END DESCRIPTION:
XS GIS Cut Line= 3
      1644455.00      6934787.99      1644205.00      6935188.00
      1644154.99      6935438.04
#Sta/Elev= 30
  4528.7 1714.54  4572.9 1712.46  4578.8 1712.93  4594.2 1712.06  4600.1 1712.25
  4609.5 1711.62  4651.9 1710.49  4870.7 1708.91  4898.4 1708.52  4919.6 1707.43
  4956.2 1706.90  4965.0 1706.43  4971.5 1704.73  4986.8 1702.08  4992.7 1701.78
  4997.5 1699.23  5003.0 1699.23  5010.6 1697.80  5047.0 1697.10  5047.5 1696.60
  5055.2 1696.60  5055.7 1697.10  5061.6 1697.98  5082.0 1702.46  5092.2 1704.04
  5143.2 1706.68  5163.6 1709.67  5184.0 1711.57  5235.0 1713.99  5255.4 1714.23
#Mann=3,-1,0
  4528.7    0.05       0  5047.0    0.03       0  5055.7    0.05       0
Bank Sta=5047,5055.7
Exp/Cntr=0.3,0.1

Type RM Length L Ch R = 1,32198,446,446,446
BEGIN DESCRIPTION:
Threemile Creek 59.0
END DESCRIPTION:
XS GIS Cut Line= 3
      1643455.00      6934938.00      1643755.00      6935238.00
      1644080.70      6935741.82
#Sta/Elev= 30
  4574.8 1717.78  4588.9 1716.99  4673.8 1714.53  4716.2 1712.29  4744.5 1712.09
  4772.8 1710.12  4786.9 1709.65  4815.2 1707.29  4829.4 1706.96  4857.6 1705.33
  4885.9 1704.74  4942.5 1704.54  4970.8 1703.98  5002.1 1702.66  5002.6 1702.16
  5010.8 1702.16  5011.3 1702.66  5064.1 1702.90  5142.6 1706.89  5215.1 1708.68
  5224.3 1708.49  5308.8 1710.12  5484.3 1710.73  5505.4 1710.40  5534.9 1710.68
  5541.7 1710.22  5547.6 1710.62  5562.8 1710.51  5593.1 1709.76  5599.0 1710.20
#Mann=3,-1,0
  4574.8    0.05       0  5002.1    0.03       0  5011.3    0.05       0
Bank Sta=5002.1,5011.3
Exp/Cntr=0.3,0.1

Type RM Length L Ch R = 1,31752,402,402,402
BEGIN DESCRIPTION:
Threemile Creek 58.0
END DESCRIPTION:
XS GIS Cut Line= 3
      1643255.00      6935238.00      1643405.00      6935488.00
      1644005.01      6936038.01
#Sta/Elev= 30
  4703.4 1715.41  4717.0 1714.66  4785.0 1713.44  4944.4 1706.69  4960.0 1705.62
  4971.6 1702.03  4981.3 1701.71  4992.0 1700.13  4998.3 1700.13  5002.0 1698.97
  5008.8 1698.42  5025.8 1698.12  5026.3 1697.62  5034.5 1697.62  5035.0 1698.12
  5051.4 1700.52  5058.8 1702.41  5079.7 1703.32  5129.7 1703.93  5228.3 1703.62
  5249.9 1704.37  5285.1 1703.51  5313.4 1704.88  5376.9 1706.46  5539.7 1708.78
  5589.7 1710.92  5709.9 1713.46  5730.9 1715.04  5738.3 1714.55  5808.9 1715.67
#Mann=3,-1,0
  4703.4    0.05       0  5025.8    0.03       0  5035.0    0.05       0
Bank Sta=5025.8,5035
Exp/Cntr=0.3,0.1

Type RM Length L Ch R = 1,31350,463,463,463
BEGIN DESCRIPTION:
Mapping XS 964b1815
END DESCRIPTION:
XS GIS Cut Line= 3
      1643117.08      6935374.25      1643110.65      6935676.44
      1643552.11      6936315.05
#Sta/Elev= 30
  4512.4 1712.48  4556.2 1711.56  4606.2 1709.66  4646.2 1709.00  4812.9 1704.01
  4934.3 1702.84  4970.1 1701.00  4976.2 1700.00  5037.2 1698.21  5037.7 1697.71
  5045.9 1697.71  5046.4 1698.21  5084.0 1700.73  5120.5 1701.76  5143.2 1701.45
  5149.3 1701.11  5156.9 1699.83  5170.2 1699.10  5179.0 1699.88  5185.1 1699.22
  5199.9 1701.21  5206.0 1701.04  5220.9 1701.92  5235.8 1701.61  5301.3 1702.67
  5358.1 1704.09  5465.6 1708.79  5531.1 1710.91  5552.1 1712.30  5591.0 1713.00
#Mann=3,-1,0
  4512.4    0.05       0  5037.2    0.03       0  5046.4    0.05       0
Bank Sta=5037.2,5046.4
Exp/Cntr=0.3,0.1

Type RM Length L Ch R = 1,30887,362,362,362
BEGIN DESCRIPTION:
Threemile Creek 57.0
END DESCRIPTION:
XS GIS Cut Line= 3
      1643104.99      6935288.04      1642905.00      6936088.00
      1642955.00      6936637.95
#Sta/Elev= 30
  4179.4 1714.71  4230.9 1713.64  4321.1 1711.04  4403.6 1708.12  4408.7 1708.23
  4468.0 1705.86  4491.2 1705.40  4550.4 1703.08  4663.8 1701.07  4692.2 1701.06
  4715.4 1700.55  4733.4 1700.80  4857.1 1700.08  4911.2 1699.03  4952.4 1699.06
  4993.7 1697.09  5006.5 1696.81  5019.2 1695.51  5019.7 1695.01  5028.4 1695.01
  5028.9 1695.51  5044.1 1696.59  5054.2 1698.69  5074.3 1700.76  5114.4 1703.21
  5174.7 1704.37  5325.3 1708.64  5345.4 1708.65  5365.5 1709.26  5556.2 1712.25
#Mann=3,-1,0
  4179.4    0.05       0  5019.2    0.03       0  5028.9    0.05       0
Bank Sta=5019.2,5028.9
Exp/Cntr=0.3,0.1

Type RM Length L Ch R = 1,30525,412,412,412
BEGIN DESCRIPTION:
Mapping XS de717e64
END DESCRIPTION:
XS GIS Cut Line= 2
      1642979.95      6935423.57      1642464.65      6936054.34
#Sta/Elev= 30
  4474.8 1709.83  4545.1 1707.91  4587.8 1706.13  4595.7 1705.41  4645.3 1703.78
  4723.5 1700.35  4765.1 1699.68  4829.2 1697.77  4865.7 1697.42  4880.0 1696.75
  4886.5 1696.01  4915.2 1695.84  4936.0 1694.49  4979.1 1694.88  4980.7 1694.47
  4981.2 1693.97  4990.0 1693.97  4990.5 1694.47  4993.5 1694.89  5022.2 1695.19
  5043.0 1699.89  5057.3 1700.83  5063.8 1700.63  5150.0 1702.45  5164.3 1702.36
  5170.8 1702.91  5191.6 1702.90  5199.5 1703.36  5220.3 1703.13  5289.3 1703.60
#Mann=3,-1,0
  4474.8    0.05       0  4980.7    0.05       0  4990.5    0.05       0
Bank Sta=4980.7,4990.5
Exp/Cntr=0.3,0.1

Type RM Length L Ch R = 1,30113,634,634,634
BEGIN DESCRIPTION:
Threemile Creek 56.0
END DESCRIPTION:
XS GIS Cut Line= 3
      1642774.20      6935250.02      1642388.50      6935520.01
      1642382.08      6935972.16
#Sta/Elev= 30
  4528.3 1710.32  4640.7 1707.45  4691.3 1706.60  4698.2 1705.86  4712.2 1705.38
  4771.5 1704.49  4828.2 1702.20  4843.0 1700.79  4849.1 1699.03  4856.9 1697.97
  4878.7 1696.22  4884.8 1695.32  4914.5 1693.87  4920.6 1692.72  4929.3 1692.71
  4935.4 1693.85  4956.3 1694.00  4965.0 1692.57  4987.2 1692.52  4987.7 1692.02
  4996.5 1692.02  4997.0 1692.52  5017.1 1693.23  5037.1 1694.72  5087.1 1696.22
  5187.1 1697.44  5227.1 1697.45  5307.1 1698.91  5327.1 1698.88  5451.3 1701.90
#Mann=3,-1,0
  4528.3    0.05       0  4987.2    0.05       0  4997.0    0.05       0
Bank Sta=4987.2,4997
Exp/Cntr=0.3,0.1

Type RM Length L Ch R = 1,29479,443,443,443
BEGIN DESCRIPTION:
Threemile Creek 55.0
END DESCRIPTION:
XS GIS Cut Line= 3
      1641705.00      6935438.00      1641855.00      6935638.00
      1642404.97      6936087.98
#Sta/Elev= 30
  4756.0 1703.67  4806.0 1702.33  4819.5 1701.49  4834.1 1701.45  4848.7 1700.42
  4892.5 1698.76  4906.0 1696.28  4913.3 1693.81  4919.5 1692.57  4927.9 1691.61
  4987.2 1687.12  4987.7 1686.62  4997.3 1686.62  4997.8 1687.12  4998.7 1687.76
  5002.9 1688.48  5009.2 1688.48  5019.6 1689.68  5027.5 1691.04  5062.7 1692.37
  5140.9 1693.21  5184.0 1694.08  5190.5 1693.86  5233.5 1694.82  5240.0 1694.61
  5254.4 1695.15  5347.0 1696.39  5538.6 1700.64  5659.9 1702.34  5716.6 1703.69
#Mann=3,-1,0
  4756.0    0.05       0  4987.2    0.03       0  4997.8    0.05       0
Bank Sta=4987.2,4997.8
Exp/Cntr=0.3,0.1

Type RM Length L Ch R = 1,29036,459,459,459
BEGIN DESCRIPTION:
Threemile Creek 54.0
END DESCRIPTION:
XS GIS Cut Line= 3
      1641555.00      6935488.03      1641555.00      6935938.00
      1641654.99      6936387.96
#Sta/Elev= 30
  4549.8 1703.24  4639.8 1701.82  4689.8 1700.64  4829.8 1696.42  4859.8 1694.74
  4889.8 1692.33  4939.8 1690.49  4969.8 1687.89  4979.8 1687.38  5004.6 1687.26
  5005.1 1686.76  5014.9 1686.76  5015.4 1687.26  5030.5 1687.71  5067.6 1687.72
  5092.0 1689.50  5111.2 1690.26  5116.3 1689.81  5159.8 1688.66  5164.9 1689.12
  5173.9 1689.03  5203.4 1690.86  5208.5 1690.49  5214.9 1691.13  5225.1 1691.42
  5245.6 1693.39  5257.1 1695.25  5300.7 1698.54  5399.3 1701.36  5460.7 1702.51
#Mann=3,-1,0
  4549.8    0.05       0  5004.6    0.03       0  5015.4    0.05       0
Bank Sta=5004.6,5015.4
Exp/Cntr=0.3,0.1

Type RM Length L Ch R = 1,28577,467,467,467
BEGIN DESCRIPTION:
Threemile Creek 53.0
END DESCRIPTION:
XS GIS Cut Line= 3
      1641354.99      6935638.03      1641155.00      6936088.00
      1641105.01      6936237.98
#Sta/Elev= 30
  4512.2 1699.07  4573.0 1697.63  4625.0 1694.42  4687.3 1692.81  4718.0 1691.71
  4723.5 1690.96  4731.0 1690.74  4741.3 1690.64  4746.8 1691.48  4775.5 1690.50
  4785.7 1690.72  4798.7 1689.96  4839.8 1689.52  4845.2 1688.75  4868.5 1688.64
  4884.2 1687.66  4915.0 1688.16  4943.7 1686.72  4967.0 1684.72  4995.7 1684.20
  4996.4 1683.83  4996.9 1683.33  5006.8 1683.33  5007.3 1683.83  5015.1 1684.68
  5036.2 1690.73  5046.8 1693.40  5057.3 1695.40  5078.4 1695.73  5162.7 1699.29
#Mann=3,-1,0
  4512.2    0.05       0  4996.4    0.05       0  5007.3    0.05       0
Bank Sta=4996.4,5007.3
Exp/Cntr=0.3,0.1

Type RM Length L Ch R = 1,28110,494,494,494
BEGIN DESCRIPTION:
Threemile Creek 52.0
END DESCRIPTION:
XS GIS Cut Line= 3
      1641204.99      6935538.00      1640805.00      6935788.00
      1640755.01      6936037.96
#Sta/Elev= 30
  4527.9 1697.83  4622.2 1694.81  4651.1 1693.21  4657.6 1692.56  4693.6 1690.83
  4797.4 1687.97  4824.5 1688.03  4846.3 1687.14  4861.0 1687.13  4882.3 1686.57
  4934.1 1684.55  4949.5 1682.84  4964.2 1682.75  4970.7 1682.18  4980.6 1681.82
  4981.1 1681.32  4991.0 1681.32  4991.5 1681.82  4996.6 1682.23  5040.4 1682.54
  5050.6 1683.90  5081.2 1690.02  5091.4 1691.49  5122.0 1693.30  5132.2 1694.41
  5152.6 1695.34  5203.6 1696.25  5213.8 1696.83  5244.3 1697.35  5254.5 1697.81
#Mann=3,-1,0
  4527.9    0.05       0  4980.6    0.05       0  4991.5    0.05       0
Bank Sta=4980.6,4991.5
Exp/Cntr=0.3,0.1

Type RM Length L Ch R = 1,27616,281,281,281
BEGIN DESCRIPTION:
Threemile Creek 51.0
END DESCRIPTION:
XS GIS Cut Line= 3
      1640555.01      6935237.99      1640455.00      6935438.00
      1640554.99      6935987.96
#Sta/Elev= 30
  4774.7 1695.62  4805.5 1693.39  4827.8 1690.29  4841.8 1689.50  4864.2 1687.12
  4878.1 1686.08  4939.6 1683.32  4953.6 1681.05  4962.0 1680.41  4984.4 1680.18
  4984.9 1679.68  4995.0 1679.68  4995.5 1680.18  5110.1 1682.20  5136.8 1683.57
  5141.9 1683.31  5190.2 1685.09  5195.2 1684.69  5221.9 1686.70  5248.6 1687.68
  5253.7 1687.34  5282.9 1688.13  5293.1 1688.94  5307.0 1689.02  5333.7 1690.06
  5354.1 1690.95  5360.4 1691.58  5404.9 1692.46  5425.2 1693.36  5557.3 1695.93
#Mann=3,-1,0
  4774.7    0.05       0  4984.4    0.05       0  4995.5    0.05       0
Bank Sta=4984.4,4995.5
Exp/Cntr=0.3,0.1

Type RM Length L Ch R = 1,27335,194,194,194
BEGIN DESCRIPTION:
Mapping XS 422c215c
END DESCRIPTION:
XS GIS Cut Line= 2
      1640162.06      6935177.17      1640363.28      6935793.66
#Sta/Elev= 30
  4799.0 1694.96  4825.4 1694.87  4831.4 1694.51  4852.0 1694.19  4873.5 1693.01
  4889.2 1691.66  4894.5 1689.90  4915.6 1686.20  4921.1 1684.49  4926.3 1684.24
  4936.6 1682.44  4978.7 1678.13  4979.2 1677.91  4979.7 1677.41  4989.9 1677.41
  4990.4 1677.91  5010.3 1678.54  5016.7 1680.26  5041.8 1681.76  5062.9 1682.44
  5080.5 1683.50  5149.6 1683.55  5240.0 1685.73  5262.7 1685.83  5309.0 1686.76
  5372.8 1687.49  5404.7 1688.04  5410.0 1688.49  5431.0 1688.76  5447.5 1689.30
#Mann=3,-1,0
  4799.0    0.05       0  4979.2    0.05       0  4990.4    0.05       0
Bank Sta=4979.2,4990.4
Exp/Cntr=0.3,0.1

Type RM Length L Ch R = 1,27141,415,415,415
BEGIN DESCRIPTION:
Threemile Creek 50.0
END DESCRIPTION:
XS GIS Cut Line= 3
      1639905.02      6935388.01      1640055.00      6935438.00
      1640404.99      6935937.99
#Sta/Elev= 30
  4840.8 1693.55  4851.3 1693.29  4861.9 1692.22  4872.4 1690.67  4882.9 1688.57
  4893.5 1684.07  4904.0 1682.55  4914.6 1682.09  4946.2 1678.73  4956.7 1677.98
  4967.3 1677.32  4982.7 1677.03  4983.2 1676.53  4993.4 1676.53  4993.9 1677.03
  5021.1 1677.90  5048.2 1681.31  5084.3 1682.91  5113.5 1683.40  5143.2 1683.31
  5185.0 1683.90  5307.1 1686.14  5315.8 1686.54  5393.4 1687.45  5487.2 1689.49
  5500.7 1690.20  5509.4 1690.06  5523.8 1690.92  5587.0 1692.55  5609.2 1693.48
#Mann=3,-1,0
  4840.8    0.05       0  4982.7    0.03       0  4993.9    0.05       0
Bank Sta=4982.7,4993.9
Exp/Cntr=0.3,0.1

Type RM Length L Ch R = 1,26726,83,83,83
BEGIN DESCRIPTION:
Mapping XS 918ed45e
END DESCRIPTION:
XS GIS Cut Line= 2
      1639574.87      6935663.57      1640221.00      6935901.06
#Sta/Elev= 30
  4751.1 1695.48  4772.6 1695.54  4815.2 1693.30  4889.4 1690.55  4919.9 1686.63
  4950.3 1679.37  4980.8 1674.44  4986.2 1674.73  5006.0 1673.64  5011.3 1674.04
  5036.4 1672.56  5041.8 1673.74  5061.3 1671.96  5061.8 1671.46  5072.1 1671.46
  5072.6 1671.96  5081.5 1673.81  5092.1 1674.07  5097.4 1675.42  5122.5 1676.26
  5127.9 1677.20  5145.4 1677.45  5158.3 1678.67  5220.0 1679.87  5244.4 1681.99
  5269.6 1685.05  5274.9 1684.68  5294.6 1685.75  5391.5 1687.25  5439.5 1689.15
#Mann=3,-1,0
  4751.1    0.05       0  5061.3    0.03       0  5072.6    0.05       0
Bank Sta=5061.3,5072.6
Exp/Cntr=0.3,0.1

Type RM Length L Ch R = 1,26643,87,87,87
BEGIN DESCRIPTION:
Threemile Creek 49.0
END DESCRIPTION:
XS GIS Cut Line= 3
      1639577.03      6935732.15      1639776.34      6935822.16
      1640149.04      6935973.37
#Sta/Elev= 30
  4785.9 1692.74  4788.6 1692.19  4857.9 1690.14  4881.0 1688.58  4886.5 1690.03
  4904.2 1688.57  4909.7 1689.46  4932.8 1688.01  4938.3 1688.83  4955.9 1688.03
  4961.4 1688.65  5004.6 1688.77  5007.7 1689.27  5031.8 1688.99  5109.4 1689.89
  5121.9 1689.56  5163.0 1690.05  5168.4 1689.56  5186.6 1689.98  5197.9 1689.19
  5229.8 1684.08  5240.4 1683.18  5240.9 1682.68  5251.2 1682.68  5251.7 1683.18
  5299.7 1684.17  5316.1 1686.44  5329.2 1687.44  5401.4 1689.49  5406.8 1690.19
#Mann=3,-1,0
  4785.9    0.05       0  5240.4    0.05       0  5251.7    0.05       0
Bank Sta=5240.4,5251.7
Exp/Cntr=0.3,0.1

Type RM Length L Ch R = 1,26556,265,265,265
BEGIN DESCRIPTION:
Mapping XS 26b4cc53
END DESCRIPTION:
XS GIS Cut Line= 2
      1639457.08      6935755.74      1640065.61      6936057.87
#Sta/Elev= 30
  4716.5 1693.67  4747.7 1693.25  4759.9 1691.86  4866.3 1688.52  4871.9 1687.29
  4888.7 1686.80  4894.3 1685.58  4933.5 1682.54  4961.5 1679.12  4983.9 1678.64
  5000.8 1679.22  5028.8 1677.71  5045.6 1679.29  5090.4 1679.87  5096.0 1678.77
  5112.8 1679.17  5118.4 1677.72  5135.2 1677.97  5143.9 1677.35  5144.4 1676.85
  5155.2 1677.35  5157.6 1678.06  5185.6 1678.40  5208.0 1680.88  5238.9 1682.62
  5283.6 1683.25  5292.1 1686.72  5305.9 1687.90  5342.5 1689.50  5395.9 1690.59
#Mann=3,-1,0
  4716.5    0.05       0  5143.9    0.05       0  5155.2    0.05       0
Bank Sta=5143.9,5155.2
Exp/Cntr=0.3,0.1

Type RM Length L Ch R = 1,26291,495,495,495
BEGIN DESCRIPTION:
Threemile Creek 48.0
END DESCRIPTION:
XS GIS Cut Line= 3
      1639404.99      6935887.98      1639555.00      6936088.00
      1639805.03      6936238.02
#Sta/Elev= 30
  4750.0 1689.76  4786.5 1687.53  4800.0 1687.31  4857.3 1683.28  4863.6 1683.38
  4886.5 1681.25  4942.7 1678.44  4957.3 1677.40  4963.6 1676.49  4978.1 1675.86
  4996.9 1673.65  5000.0 1673.65  5002.1 1673.00  5002.6 1672.50  5012.9 1672.50
  5013.4 1673.00  5013.6 1673.27  5023.3 1673.47  5035.0 1675.19  5044.7 1676.15
  5058.3 1676.80  5081.7 1676.76  5108.9 1675.27  5116.6 1675.22  5161.3 1678.64
  5182.7 1680.90  5188.6 1682.25  5219.7 1685.96  5278.0 1688.54  5291.6 1688.83
#Mann=3,-1,0
  4750.0    0.05       0  5002.1    0.03       0  5013.4    0.05       0
Bank Sta=5002.1,5013.4
Exp/Cntr=0.3,0.1

Type RM Length L Ch R = 1,25796,474,474,474
BEGIN DESCRIPTION:
Threemile Creek 47.0
END DESCRIPTION:
XS GIS Cut Line= 3
      1639024.18      6936175.71      1639205.00      6936438.00
      1639405.02      6936588.01
#Sta/Elev= 30
  4681.8 1683.93  4721.0 1683.24  4727.2 1682.86  4748.2 1683.00  4798.9 1680.30
  4849.6 1676.97  4855.7 1677.13  4885.4 1676.06  4942.2 1675.09  4951.0 1674.44
  4957.1 1674.69  4992.9 1672.53  4997.3 1671.65  5003.5 1671.65  5013.9 1670.60
  5037.4 1669.68  5037.9 1669.18  5048.2 1669.18  5048.7 1669.68  5057.7 1670.63
  5063.9 1672.33  5078.5 1674.54  5107.7 1677.23  5128.5 1680.72  5143.1 1682.44
  5157.7 1683.24  5163.9 1684.05  5200.4 1685.45  5207.7 1686.08  5250.4 1687.43
#Mann=3,-1,0
  4681.8    0.05       0  5037.4    0.03       0  5048.7    0.05       0
Bank Sta=5037.4,5048.7
Exp/Cntr=0.3,0.1

Type RM Length L Ch R = 1,25322,416,416,416
BEGIN DESCRIPTION:
Threemile Creek 46.0
END DESCRIPTION:
XS GIS Cut Line= 3
      1638707.04      6936227.15      1638805.00      6936638.00
      1638916.70      6936843.66
#Sta/Elev= 30
  4572.9 1679.51  4676.8 1680.07  4755.9 1678.59  4761.0 1678.77  4803.2 1677.31
  4830.8 1675.73  4882.2 1673.99  4887.4 1673.43  4943.9 1671.61  4971.6 1670.11
  4992.7 1669.57  5009.0 1669.76  5012.3 1669.19  5012.8 1668.69  5023.2 1668.69
  5023.7 1669.19  5025.2 1669.56  5040.8 1669.20  5052.8 1669.65  5068.9 1672.78
  5074.9 1674.58  5085.1 1676.24  5090.8 1676.61  5097.7 1678.23  5106.9 1678.96
  5112.6 1678.81  5150.7 1681.53  5172.5 1681.44  5188.7 1682.06  5229.3 1682.54
#Mann=3,-1,0
  4572.9    0.05       0  5012.3    0.03       0  5023.7    0.05       0
Bank Sta=5012.3,5023.7
Exp/Cntr=0.3,0.1

Type RM Length L Ch R = 1,24906,482,482,482
BEGIN DESCRIPTION:
Threemile Creek 45.0
END DESCRIPTION:
XS GIS Cut Line= 3
      1638177.75      6936400.73      1638488.47      6936863.60
      1638786.36      6936867.88
#Sta/Elev= 30
  4535.6 1682.03  4568.4 1680.58  4640.7 1679.38  4668.0 1678.13  4683.0 1678.07
  4755.0 1674.78  4770.0 1674.67  4791.0 1673.12  4806.0 1672.84  4827.0 1671.39
  4842.0 1671.18  4863.1 1669.96  4905.7 1669.31  4920.1 1669.66  5001.3 1667.75
  5001.8 1667.25  5012.3 1667.25  5012.8 1667.75  5022.1 1669.52  5058.1 1673.12
  5064.1 1673.02  5073.1 1673.83  5079.1 1673.65  5086.3 1674.36  5099.6 1674.12
  5169.6 1676.02  5229.6 1676.99  5289.6 1679.22  5339.6 1679.75  5391.0 1681.30
#Mann=3,-1,0
  4535.6    0.05       0  5001.3    0.05       0  5012.8    0.05       0
Bank Sta=5001.3,5012.8
Exp/Cntr=0.3,0.1

Type RM Length L Ch R = 1,24424,443,443,443
BEGIN DESCRIPTION:
Threemile Creek 44.0
END DESCRIPTION:
XS GIS Cut Line= 3
      1638205.00      6937138.00      1638305.00      6937088.00
      1638704.98      6936888.01
#Sta/Elev= 30
  4887.9 1681.13  4901.9 1679.62  4932.6 1678.29  4941.0 1676.63  4946.6 1674.88
  4955.0 1670.34  4963.4 1666.49  4969.0 1665.29  4991.1 1663.39  4991.6 1662.89
  5002.2 1662.89  5002.7 1663.39  5022.1 1663.85  5030.5 1664.72  5044.4 1667.46
  5058.4 1669.00  5075.2 1669.40  5097.5 1670.96  5111.5 1670.96  5119.9 1670.33
  5178.6 1671.60  5201.0 1671.59  5237.3 1672.96  5276.4 1673.44  5298.8 1674.18
  5304.4 1674.76  5321.1 1674.95  5365.9 1677.68  5388.2 1677.86  5446.9 1679.68
#Mann=3,-1,0
  4887.9    0.05       0  4991.1    0.03       0  5002.7    0.05       0
Bank Sta=4991.1,5002.7
Exp/Cntr=0.3,0.1

Type RM Length L Ch R = 1,23981,501,501,501
BEGIN DESCRIPTION:
Threemile Creek 43.0
END DESCRIPTION:
XS GIS Cut Line= 3
      1638505.00      6937438.00      1638637.76      6937368.60
      1638910.31      6937198.08
#Sta/Elev= 30
  4850.2 1676.28  4880.5 1675.15  4886.1 1674.06  4924.6 1669.96  4940.5 1668.94
  4952.4 1665.69  4963.0 1664.78  4968.8 1663.63  4974.4 1660.70  4985.1 1659.94
  4985.6 1659.44  4996.2 1659.44  4996.7 1659.94  5020.3 1661.29  5033.7 1663.55
  5070.3 1666.13  5100.9 1666.82  5106.8 1667.39  5114.7 1667.09  5158.7 1668.26
  5173.7 1669.28  5201.1 1669.91  5222.4 1671.05  5244.5 1672.97  5268.1 1673.84
  5274.2 1674.91  5280.1 1674.66  5295.5 1675.44  5316.7 1677.04  5321.5 1677.86
#Mann=3,-1,0
  4850.2    0.05       0  4985.1    0.03       0  4996.7    0.05       0
Bank Sta=4985.1,4996.7
Exp/Cntr=0.3,0.1

Type RM Length L Ch R = 1,23480,469,469,469
BEGIN DESCRIPTION:
Threemile Creek 42.0
END DESCRIPTION:
XS GIS Cut Line= 3
      1638505.00      6937638.00      1638905.00      6937738.00
      1639054.99      6937738.00
#Sta/Elev= 30
  4587.3 1676.46  4669.8 1673.31  4721.3 1670.29  4729.0 1669.92  4734.2 1670.17
  4770.3 1667.79  4803.8 1667.11  4816.6 1666.44  4875.9 1665.77  4906.8 1664.95
  4927.5 1663.82  4948.1 1663.53  4968.7 1662.20  4981.6 1661.77  4989.3 1661.12
  4997.0 1659.83  5002.1 1659.83  5003.8 1659.04  5004.3 1658.54  5015.0 1658.54
  5015.5 1659.04  5029.6 1659.86  5039.6 1661.80  5049.6 1664.20  5069.6 1666.93
  5089.6 1668.82  5109.6 1672.48  5129.6 1677.26  5147.1 1680.17  5149.6 1680.17
#Mann=3,-1,0
  4587.3    0.05       0  5003.8    0.05       0  5015.5    0.05       0
Bank Sta=5003.8,5015.5
Exp/Cntr=0.3,0.1

Type RM Length L Ch R = 1,23011,441,441,441
BEGIN DESCRIPTION:
Threemile Creek 41.0
END DESCRIPTION:
XS GIS Cut Line= 3
      1638455.01      6937838.01      1638705.00      6938138.00
      1638805.00      6938188.00
#Sta/Elev= 30
  4610.0 1673.28  4631.5 1671.91  4680.9 1669.79  4695.2 1668.55  4716.1 1667.57
  4734.0 1667.56  4738.4 1667.55  4744.7 1666.42  4773.4 1665.21  4865.8 1663.21
  4872.3 1663.61  4880.1 1663.46  4936.1 1661.55  4943.9 1661.19  4964.7 1658.62
  4979.0 1657.56  4997.2 1656.54  5017.0 1656.17  5017.5 1655.67  5028.2 1655.67
  5028.7 1656.17  5031.2 1656.89  5045.2 1658.25  5053.6 1661.86  5067.6 1666.59
  5076.0 1668.34  5081.6 1670.42  5089.9 1672.48  5098.3 1674.01  5112.3 1674.91
#Mann=5,-1,0
  4610.0    0.05       0  4734.0    0.12       0  4738.4    0.05       0
  5017.0    0.05       0  5028.7    0.05       0
Bank Sta=5017,5028.7
Exp/Cntr=0.3,0.1

Type RM Length L Ch R = 1,22570,446,446,446
BEGIN DESCRIPTION:
Threemile Creek 40.0
END DESCRIPTION:
XS GIS Cut Line= 3
      1638205.01      6937988.01      1638355.00      6938388.00
      1638554.97      6938637.97
#Sta/Elev= 30
  4577.0 1670.54  4666.3 1666.15  4719.6 1664.36  4854.7 1660.91  4886.7 1660.65
  4918.7 1659.37  4933.9 1658.68  4940.1 1656.80  4958.8 1654.50  4976.7 1653.72
  4977.2 1653.22  4988.4 1653.22  4988.9 1653.72  4994.4 1654.56  5007.4 1654.38
  5011.4 1655.16  5032.2 1656.49  5068.2 1656.90  5075.4 1657.98  5089.8 1658.81
  5096.2 1661.50  5104.2 1663.28  5110.6 1663.80  5132.2 1664.51  5160.3 1662.97
  5168.3 1663.27  5174.7 1663.83  5182.7 1665.62  5260.3 1669.88  5324.3 1674.59
#Mann=5,-1,0
  4577.0    0.05       0  4666.3    0.12       0  4719.6    0.05       0
  4976.7    0.03       0  4988.9    0.05       0
Bank Sta=4976.7,4988.9
Exp/Cntr=0.3,0.1

Type RM Length L Ch R = 1,22124,485,485,485
BEGIN DESCRIPTION:
Threemile Creek 39.0
END DESCRIPTION:
XS GIS Cut Line= 3
      1637704.98      6938087.96      1637955.00      6938488.00
      1638004.98      6938587.96
#Sta/Elev= 30
  4527.7 1674.89  4556.6 1673.89  4577.9 1671.95  4586.7 1670.51  4724.1 1661.34
  4818.4 1657.97  4839.7 1656.86  4846.1 1657.10  4891.5 1655.60  4905.1 1654.20
  4912.8 1652.97  4918.7 1654.12  4934.0 1655.90  4949.3 1654.57  4955.2 1654.80
  4964.1 1654.08  4970.5 1651.83  4990.4 1649.75  4990.9 1649.25  5002.1 1649.25
  5002.6 1649.75  5013.4 1651.15  5021.8 1653.48  5035.8 1654.70  5052.5 1658.77
  5058.1 1659.04  5080.5 1663.40  5097.3 1667.55  5108.4 1669.50  5111.2 1669.50
#Mann=3,-1,0
  4527.7    0.05       0  4990.4    0.05       0  5002.6    0.05       0
Bank Sta=4990.4,5002.6
Exp/Cntr=0.3,0.1

Type RM Length L Ch R = 1,21639,270,270,270
BEGIN DESCRIPTION:
Threemile Creek 38.0
END DESCRIPTION:
XS GIS Cut Line= 3
      1637355.00      6938438.00      1637505.00      6938588.00
      1637804.96      6938737.98
#Sta/Elev= 30
  4794.7 1670.55  4798.2 1670.55  4823.0 1666.82  4837.1 1663.62  4851.3 1661.35
  4879.6 1658.04  4893.7 1657.01  4907.8 1656.58  4950.3 1653.18  4964.4 1651.90
  4972.4 1650.14  4972.9 1649.64  4984.1 1649.64  4984.6 1650.14  5003.3 1652.16
  5029.2 1652.21  5065.5 1651.13  5082.3 1652.35  5087.9 1653.22  5127.0 1653.95
  5149.4 1654.92  5155.0 1655.90  5194.1 1658.24  5199.7 1659.86  5216.5 1661.05
  5222.1 1662.23  5230.4 1663.26  5319.9 1667.66  5328.3 1668.70  5342.2 1668.94
#Mann=3,-1,0
  4794.7    0.05       0  4972.4    0.03       0  4984.6    0.05       0
Bank Sta=4972.4,4984.6
Exp/Cntr=0.3,0.1

Type RM Length L Ch R = 1,21369,283,283,283
BEGIN DESCRIPTION:
Mapping XS dda8f528
END DESCRIPTION:
XS GIS Cut Line= 3
      1637140.63      6938655.05      1637517.75      6938884.32
      1637610.99      6938877.97
#Sta/Elev= 30
  4819.7 1669.54  4848.2 1668.94  4860.0 1667.54  4869.6 1666.11  4875.5 1663.74
  4906.4 1657.78  4918.4 1655.66  4933.6 1654.30  4955.0 1650.64  4964.3 1648.35
  4964.8 1647.85  4976.0 1647.85  4976.5 1648.35  4985.9 1649.03  4991.8 1648.95
  5000.4 1650.06  5013.1 1650.69  5022.7 1650.68  5028.6 1650.04  5044.0 1650.35
  5058.9 1651.20  5065.4 1651.87  5071.2 1653.09  5108.0 1654.86  5152.5 1654.30
  5224.3 1655.36  5233.9 1656.13  5276.9 1656.69  5318.4 1658.46  5354.5 1660.59
#Mann=3,-1,0
  4819.7    0.05       0  4964.3    0.03       0  4976.5    0.05       0
Bank Sta=4964.3,4976.5
Exp/Cntr=0.3,0.1
