HEC-RAS study Buck Creek.prj: Buck Creek Base Level Engineering

--- Buck Creek.g01 (geometry) --- (continued)

Type RM Length L Ch R = 1 ,66021   ,507,507,507
BEGIN DESCRIPTION:
Buck Creek 66020.61
END DESCRIPTION:
XS GIS Cut Line= 3
      1630895.49      6841463.51        1631195.      6841789.06
      1631517.92      6842447.91
#Sta/Elev= 30
  4561.6 1877.32  4571.4 1877.22  4621.3 1873.12  4734.1 1867.03  4755.7 1864.96
    4805 1862.69  4812.3 1861.61  4840.2 1860.93  4868.5 1857.55  4875.9 1859.58
  4891.1 1860.78  4904.3 1861.15  4911.1 1862.69  4918.5 1862.16  4932.7 1860.16
  4939.4 1858.54  4946.8 1855.68  4954.6 1855.15  4955.1 1854.65  4967.4 1855.15
  4988.9  1855.5  5000.3  1857.8  5006.2  1857.8  5011.8 1860.23  5025.1  1862.4
  5064.5 1863.56  5079.3 1864.36  5169.3 1863.24  5303.5 1863.73  5737.7 1869.85
#Mann= 5 ,-1 , 0
  4561.6     .05       0  4891.1     .12       0  4954.6     .07       0
  4967.4     .12       0  5064.5     .05       0
Bank Sta=4954.6,4967.4
XS Rating Curve= 0 ,0
Exp/Cntr=0.3,0.1

Type RM Length L Ch R = 1 ,65514   ,702,702,702
BEGIN DESCRIPTION:
Buck Creek 65514.36
END DESCRIPTION:
XS GIS Cut Line= 3
      1630606.45      6841473.93      1630715.84      6841880.21
      1630908.54      6842557.28
#Sta/Elev= 30
  4582.8 1873.88  4594.3  1873.4  4607.7 1873.37  4618.1 1872.23  4634.3 1868.14
  4639.4 1868.49    4669 1865.31  4674.2 1865.69  4700.9 1863.09  4742.4 1861.67
  4788.9 1861.02  4845.9 1859.62  4928.8 1859.55  4938.3 1859.89  4943.5 1860.49
  4959.8 1858.63  4971.8 1854.31  4972.3 1853.81  4984.2 1853.81  4984.7 1854.31
  4990.9 1856.42  5003.5 1856.69  5017.8 1857.71  5056.9 1858.63  5105.2 1857.59
  5197.5 1861.43  5314.7 1862.06  5416.3 1863.36  5460.5 1863.37  5707.5  1866.6
#Mann= 3 ,-1 , 0
  4582.8     .05       0  4971.8     .03       0  4984.7     .05       0
Bank Sta=4971.8,4984.7
XS Rating Curve= 0 ,0
Exp/Cntr=0.3,0.1

Type RM Length L Ch R = 1 ,64812   ,513,513,513
BEGIN DESCRIPTION:
Buck Creek 64811.98
END DESCRIPTION:
XS GIS Cut Line= 3
       1630344.3      6841527.82      1630224.52      6842087.67
      1630146.55      6842724.39
#Sta/Elev= 30
  4427.4 1862.45  4450.5 1861.01  4570.8 1857.66  4643.3 1856.55    4673 1856.59
  4693.5 1855.88  4765.1 1856.47  4775.3 1856.31  4786.6 1855.19  4795.7 1855.03
  4969.1 1855.09  4974.2 1854.96  4979.8 1853.84  5002.6 1853.65  5003.8  1852.6
  5004.3  1852.1  5016.3  1852.1  5016.8  1852.6  5030.5  1854.5  5036.3 1855.94
  5041.3  1855.6  5060.7 1858.93  5080.8 1860.26  5204.2 1861.44  5367.1 1864.11
  5383.1  1865.1  5483.8 1867.21  5524.1 1868.86    5530 1869.44  5641.4 1872.17
#Mann= 3 ,-1 , 0
  4427.4     .05       0  5003.8     .05       0  5016.8     .05       0
Bank Sta=5003.8,5016.8
XS Rating Curve= 0 ,0
Exp/Cntr=0.3,0.1

Type RM Length L Ch R = 1 ,64299   ,307,307,307
BEGIN DESCRIPTION:
Buck Creek 64298.97
END DESCRIPTION:
XS GIS Cut Line= 4
       1629841.5      6841528.88      1629721.91      6842006.95
       1629711.5      6842087.67      1629734.93      6842699.63
#Sta/Elev= 30
  4425.8 1861.35  4445.5 1860.69  4472.2 1856.36  4486.7 1855.59    4497 1856.81
  4518.6 1856.58    4528 1854.33  4683.5 1853.61  4703.2 1852.49  4724.7 1853.59
  4760.7 1852.44  4765.9 1853.94    4802 1852.07  4807.1 1852.87  4848.4 1849.76
  4884.4 1849.41  4889.6 1847.79  4927.7 1847.42  4928.2 1846.92  4940.7 1847.42
  4980.2 1848.25  5030.3 1854.43  5048.9 1854.93  5058.2  1855.3  5122.5 1857.26
  5240.5 1862.46  5390.6 1866.67  5450.6 1869.96  5540.7 1872.37  5612.4 1872.67
#Mann= 7 ,-1 , 0
  4425.8     .05       0  4760.7     .12       0  4927.7     .07       0
  4940.7     .12       0  5048.9     .05       0  5058.2     .12       0
  5122.5     .05       0
Bank Sta=4927.7,4940.7
XS Rating Curve= 0 ,0
Exp/Cntr=0.3,0.1

Type RM Length L Ch R = 1 ,63992   ,355,355,355
BEGIN DESCRIPTION:
Buck Creek 63992.1
END DESCRIPTION:
XS GIS Cut Line= 4
       1629469.1      6841614.84      1629445.87      6842030.38
       1629461.5      6842189.24      1629508.37      6842697.07
#Sta/Elev= 30
    4425 1856.91  4448.2 1855.75  4468.2  1853.1  4478.2 1853.03  4488.3 1854.19
  4508.3    1854  4518.3 1852.25  4528.3 1853.12  4558.4 1853.81  4765.4 1854.14
  4883.7 1853.11  4899.1 1852.66  4926.5 1850.17  4939.3 1850.18  4949.3 1851.46
  4959.4 1851.39  5013.1 1847.69  5013.6 1847.19  5025.7 1847.19  5026.2 1847.69
  5029.7 1848.98  5049.3 1852.14  5059.8 1853.37  5089.1  1859.6  5140.2 1860.91
  5150.2 1862.15  5220.5 1863.48    5341 1867.95  5411.3 1869.48  5510.8 1868.89
#Mann= 5 ,-1 , 0
    4425     .05       0  4926.5     .12       0  5013.1     .07       0
  5026.2     .12       0  5049.3     .05       0
Bank Sta=5013.1,5026.2
XS Rating Curve= 0 ,0
Exp/Cntr=0.3,0.1

Type RM Length L Ch R = 1 ,63637   ,179,179,179
BEGIN DESCRIPTION:
Buck Creek 63637.04
END DESCRIPTION:
XS GIS Cut Line= 4
      1628867.74      6841131.94      1629083.89      6841999.13
      1629107.33      6842186.63      1629104.73      6842449.64
#Sta/Elev= 30
  3920.8 1866.67  4030.1 1859.79  4081.6 1858.69  4178.9 1851.78    4195 1852.54
  4287.8 1850.69  4370.2 1851.49  4390.8 1850.57  4411.4 1854.54  4442.3 1855.59
  4483.6 1852.89  4535.1 1853.86  4576.3 1849.47  4607.2 1851.58  4873.8 1850.02
  4914.2 1852.51  4924.2 1851.84  4941.9 1846.68  4946.9 1847.48  4964.5 1841.68
  4978.2 1840.98  4978.7 1840.48  4991.3 1840.98  5006.7  1841.2  5024.9  1850.1
  5034.9 1853.27  5064.9 1856.22  5134.9 1858.82  5204.9  1859.1  5266.5 1861.19
#Mann= 3 ,-1 , 0
  3920.8     .05       0  4978.2     .03       0  4991.3     .05       0
Bank Sta=4978.2,4991.3
XS Rating Curve= 0 ,0
Exp/Cntr=0.3,0.1

Type RM Length L Ch R = 1 ,63458   ,653,653,653
BEGIN DESCRIPTION:
Buck Creek 63457.53
END DESCRIPTION:
XS GIS Cut Line= 4
      1628698.46      6841165.76      1628914.62      6841952.26
      1628943.27      6842144.97      1628945.86      6842424.57
#Sta/Elev= 30
  3996.1 1866.43  4042.4 1865.29  4133.2 1858.26  4205.8 1856.37  4247.3 1852.92
  4288.8 1853.44  4423.6 1850.32  4444.4 1850.84  4457.3 1849.55  4465.1 1849.59
  4491.7  1853.7  4531.4 1854.31  4558.4 1852.21  4599.9 1853.87    4631 1852.43
  4651.8 1849.34  4662.2    1849  4703.6 1851.39  4837.8 1848.25    4920  1849.2
  4938.9 1847.98  4942.4 1846.05  4942.9 1845.55  4955.5 1846.05  4969.2 1847.84
  4999.5 1846.18  5039.6  1847.2  5089.6 1852.69  5129.6  1855.1  5286.2 1858.13
#Mann= 3 ,-1 , 0
  3996.1     .05       0  4942.4     .03       0  4955.5     .05       0
Bank Sta=4942.4,4955.5
XS Rating Curve= 0 ,0
Exp/Cntr=0.3,0.1

Type RM Length L Ch R = 1 ,62805   ,454,454,454
BEGIN DESCRIPTION:
Buck Creek 62805.2
END DESCRIPTION:
XS GIS Cut Line= 3
      1627810.46      6841522.57      1628307.85      6842194.45
      1628859.89      6842462.66
#Sta/Elev= 30
  4167.2 1864.86  4246.4 1863.65  4352.8 1857.55  4388.3 1857.75  4402.9 1856.65
  4417.6 1853.56  4460.1 1852.77  4509.9 1848.64  4559.7  1851.5  4603.3 1849.59
  4653.4 1851.72  4674.2 1850.98  4703.5  1846.1  4732.7 1845.13  4759.8 1845.92
  4789.1 1849.65  4818.3 1849.68  4839.2 1848.83  4853.8 1842.66  4945.6  1845.5
  4968.6 1842.35  4988.9 1841.97  4989.4 1841.47  5002.4 1841.97  5019.7 1842.62
  5047.8 1846.09  5087.4 1845.57    5155 1847.43  5256.4 1853.93  5616.9 1856.88
#Mann= 3 ,-1 , 0
  4167.2     .05       0  4988.9     .03       0  5002.4     .05       0
Bank Sta=4988.9,5002.4
XS Rating Curve= 0 ,0
Exp/Cntr=0.3,0.1

Type RM Length L Ch R = 1 ,62351   ,366,366,366
BEGIN DESCRIPTION:
Buck Creek 62351.01
END DESCRIPTION:
XS GIS Cut Line= 3
      1627592.98      6842564.76      1628199.78      6842538.72
      1628710.14      6842465.81
#Sta/Elev= 30
  4396.1 1855.86  4418.1 1854.77  4428.1 1855.11  4435.1 1854.01  4440.1 1854.25
  4538.2 1850.73  4638.3 1841.31  4666.8 1839.65  4698.4 1840.58  4748.4 1843.34
  4798.5 1843.49  4868.6  1842.8  4918.6 1841.58  4978.7 1838.93  4981.9 1836.87
  4982.4 1836.37    4995 1836.37  4995.5 1836.87  4998.6 1838.13  5003.5 1838.13
  5008.7  1840.1  5038.9 1845.36  5150.1 1844.78  5210.8 1845.83  5241.1 1846.74
  5326.8 1850.98  5372.4 1854.52  5453.2 1855.11  5463.2 1855.74    5519 1855.53
#Mann= 3 ,-1 , 0
  4396.1     .05       0  4981.9     .05       0  4995.5     .05       0
Bank Sta=4981.9,4995.5
XS Rating Curve= 0 ,0
Exp/Cntr=0.3,0.1

Type RM Length L Ch R = 1 ,61985   ,337,337,337
BEGIN DESCRIPTION:
Buck Creek 61984.8
END DESCRIPTION:
XS GIS Cut Line= 3
      1627553.96      6842788.72      1628012.28      6842835.59
      1628721.59      6842635.53
#Sta/Elev= 30
  4540.1 1858.18  4571.3 1858.32  4651.7 1854.03    4702 1852.76  4778.1 1849.47
  4802.5 1849.25  4842.7 1847.52  4872.5 1845.26  4877.5  1845.9  4882.9 1844.38
  4923.1 1840.38  4943.2 1836.26  4963.3 1836.97  4970.1 1835.67  4970.6 1835.17
  4983.7 1835.67  4993.5 1836.46  4999.7 1838.11  5004.8 1838.11  5009.6 1839.34
  5014.8 1838.19  5034.8 1841.42  5082.8 1843.31    5088 1842.86  5097.2  1843.7
  5336.1 1843.54    5440 1844.79  5512.8 1846.77  5606.3 1852.91  5737.8 1855.05
#Mann= 3 ,-1 , 0
  4540.1     .05       0  4970.1     .05       0  4983.7     .05       0
Bank Sta=4970.1,4983.7
XS Rating Curve= 0 ,0
Exp/Cntr=0.3,0.1

Type RM Length L Ch R = 1 ,61648   ,309,309,309
BEGIN DESCRIPTION:
Buck Creek 61647.98
END DESCRIPTION:
XS GIS Cut Line= 3
      1627698.52      6843278.29      1628099.95      6843141.58
      1628920.16      6842768.37
#Sta/Elev= 30
  4574.3 1857.72  4619.9 1855.53  4697.4 1853.24    4714 1851.93  4739.6 1851.43
  4771.3 1849.51  4776.7 1848.47  4855.8 1845.39  4902.1 1841.96  4950.9 1836.13
  4975.8 1834.81  4976.3 1834.31  4988.9 1834.31  4989.4 1834.81  4990.9 1835.56
  4998.4 1835.32  5003.9  1836.9  5019.7 1837.65  5048.3 1841.49  5080.8 1840.76
  5209.7 1842.21  5322.5 1842.24  5520.3  1843.9  5595.1 1845.36  5663.4 1848.34
    5804 1855.21  5819.1 1856.19  5842.2 1856.22  5849.9 1856.92  5899.5 1857.96
#Mann= 5 ,-1 , 0
  4574.3     .05       0  4975.8     .05       0  4989.4     .05       0
  5663.4     .12       0    5804     .05       0
Bank Sta=4975.8,4989.4
XS Rating Curve= 0 ,0
Exp/Cntr=0.3,0.1

Type RM Length L Ch R = 1 ,61339   ,278,278,278
BEGIN DESCRIPTION:
Buck Creek 61339.01
END DESCRIPTION:
XS GIS Cut Line= 3
      1627883.42      6843572.31      1628188.96      6843423.01
      1629067.48      6842926.46
#Sta/Elev= 30
  4660.3 1854.35  4685.7 1853.85  4725.2 1851.71  4753.3 1850.96  4770.2 1849.09
  4888.4 1842.66  4927.8 1837.63  4950.4 1835.82  4978.4  1835.1  5000.4 1835.49
    5010 1834.81  5010.5 1834.31  5023.2 1834.31  5023.7 1834.81  5038.5 1837.46
  5044.3 1837.81  5060.2 1840.31  5097.7 1839.85  5221.9 1841.62  5432.6 1841.94
  5647.8 1843.76  5765.4  1846.2  5777.7 1847.34  5815.2 1848.03  5852.8 1850.59
  5858.5 1851.66  5870.4 1852.64  5955.3 1855.03  5971.2 1856.52  6009.5 1856.16
#Mann= 4 ,-1 , 0
  4660.3     .05       0    5010     .05       0  5023.7     .05       0
  5870.4     .12       0
Bank Sta=5010,5023.7
XS Rating Curve= 0 ,0
Exp/Cntr=0.3,0.1

Type RM Length L Ch R = 1 ,61061   ,260,260,260
BEGIN DESCRIPTION:
Buck Creek 61060.69
END DESCRIPTION:
XS GIS Cut Line= 3
      1627869.48      6843811.91      1628254.93      6843683.43
      1629254.97      6843120.91
#Sta/Elev= 30
  4590.1 1858.37  4683.5 1855.81  4796.2 1850.64  4817.3  1848.8  4859.4 1847.14
  4904.9 1844.08  4922.7 1841.54  4936.5 1839.02  4943.8 1837.15  4962.9 1835.16
  5030.5 1833.52    5031 1833.02  5043.7 1833.02  5044.2 1833.52  5065.3 1838.08
  5080.7 1839.57  5096.6 1838.18  5183.3 1839.81    5205 1839.88  5258.5 1838.73
  5485.5  1841.8  5765.2 1844.29  5911.9 1846.91  5976.9 1849.23  5983.2 1850.67
  5992.8 1850.79  5998.6 1851.57  6014.5 1850.93  6073.8 1853.89  6143.8 1856.12
#Mann= 3 ,-1 , 0
  4590.1     .05       0  5030.5     .05       0  5044.2     .05       0
Bank Sta=5030.5,5044.2
XS Rating Curve= 0 ,0
Exp/Cntr=0.3,0.1

Type RM Length L Ch R = 1 ,60801   ,270,270,270
BEGIN DESCRIPTION:
Buck Creek 60801.45
END DESCRIPTION:
XS GIS Cut Line= 3
      1628025.79      6844082.72      1628404.24      6843888.29
       1629470.1      6843440.42
#Sta/Elev= 30
  4579.3 1859.15  4670.1 1857.32  4819.8 1850.69  4848.2 1848.15  4893.2  1845.4
  4908.5 1843.53  4925.1 1841.11  4947.2 1836.24  4952.9 1834.19  4976.2 1830.91
  4976.7 1830.41  4989.5 1830.41    4990 1830.91  5002.4  1833.3  5007.9  1833.3
  5020.1 1836.15  5038.1 1836.74  5049.3 1838.17  5067.7  1837.6  5157.5 1839.12
  5461.9 1840.39    5922 1847.17  5945.8 1848.91  5960.1 1848.34  5998.7  1850.3
  6004.1 1849.96  6022.5  1851.3  6080.8 1853.29  6099.2 1854.76  6160.9 1855.99
#Mann= 3 ,-1 , 0
  4579.3     .05       0  4976.2     .05       0    4990     .05       0
Bank Sta=4976.2,4990
XS Rating Curve= 0 ,0
Exp/Cntr=0.3,0.1

Type RM Length L Ch R = 1 ,60531   ,300,300,300
BEGIN DESCRIPTION:
Buck Creek 60530.9
END DESCRIPTION:
XS GIS Cut Line= 3
      1628112.59      6844266.76      1628553.55      6844103.57
      1629556.98      6843798.02
#Sta/Elev= 30
  4530.2 1855.16  4634.2 1853.34  4655.8 1852.69  4661.2 1853.04  4741.7 1849.88
  4802.5 1848.52  4895.3 1844.78  4918.8 1841.55  4967.3 1829.61  4967.8 1829.11
  4980.6 1829.11  4981.1 1829.61  5004.7 1831.12  5022.5 1834.45  5051.8 1837.06
  5381.7 1839.01    5584  1841.7  5702.3 1843.93  5785.9 1847.88  5791.5 1848.82
  5824.4  1851.6  5857.2  1854.1  5862.4 1853.92  5869.5 1855.43    5880 1856.01
  5933.4 1857.29    5961 1858.97  5966.2 1858.74  5993.8  1860.3  6049.3 1862.23
#Mann= 6 ,-1 , 0
  4530.2     .12       0  4634.2     .05       0  4967.3     .05       0
  4981.1     .05       0  5022.5     .12       0  5051.8     .05       0
Bank Sta=4967.3,4981.1
XS Rating Curve= 0 ,0
Exp/Cntr=0.3,0.1

Type RM Length L Ch R = 1 ,60231   ,444,444,444
BEGIN DESCRIPTION:
Buck Creek 60230.62
END DESCRIPTION:
XS GIS Cut Line= 3
      1628334.86      6844478.82      1628704.62      6844346.88
      1629423.34      6844162.86
#Sta/Elev= 30
  4607.1 1841.83  4629.1 1840.37  4649.3 1838.15  4654.6 1838.98  4660.3 1837.94
  4680.1 1836.61  4685.4 1837.13  4692.2 1836.41  4746.8 1836.11  4852.9 1836.65
  4915.2 1836.92  4946.7 1835.82    4952 1835.46  4957.6 1833.51  4977.5 1829.32
  4990.3 1828.17  4990.8 1827.67  5003.6 1827.67  5004.1 1828.17  5031.1    1829
  5054.9 1834.62    5062 1836.59  5103.3 1835.88  5178.7 1836.43  5309.8 1838.45
    5413 1839.14  5588.5 1842.26  5640.1 1845.27  5698.8 1851.79  5741.6  1854.4
#Mann= 6 ,-1 , 0
  4607.1     .12       0  4746.8     .05       0  4852.9     .12       0
  4990.3     .07       0  5004.1     .12       0  5054.9     .05       0
Bank Sta=4990.3,5004.1
XS Rating Curve= 0 ,0
Exp/Cntr=0.3,0.1

Type RM Length L Ch R = 1 ,59787   ,359,359,359
BEGIN DESCRIPTION:
Buck Creek 59787.38
END DESCRIPTION:
XS GIS Cut Line= 3
      1628352.24       6844544.8      1629048.37      6844584.73
      1629525.81      6844378.13
#Sta/Elev= 30
  4304.6 1834.77  4415.6 1834.95  4514.6 1835.49  4613.6 1835.46  4647.9  1834.5
    4718 1834.34  4768.1 1835.26  4818.2 1834.56  4838.2 1832.89  4868.3 1833.61
  4878.3  1833.3  4901.4 1829.29  4901.9 1828.79  4914.8 1828.79  4915.3 1829.29
  4918.4 1832.28  4928.4  1833.8  5010.4 1832.48  5033.9  1834.5  5041.8 1837.19
  5057.4 1838.55  5086.3 1838.81  5104.3 1839.72  5261.6 1840.71    5361 1843.21
  5401.4 1845.58  5431.5 1849.27  5466.7 1852.27  5507.4 1854.17  5522.1 1854.17
#Mann= 6 ,-1 , 0
  4304.6     .12       0  4415.6     .05       0  4514.6     .12       0
  4613.6     .05       0  4901.4     .05       0  4915.3     .05       0
Bank Sta=4901.4,4915.3
XS Rating Curve= 0 ,0
Exp/Cntr=0.3,0.1

Type RM Length L Ch R = 1 ,59428   ,386,386,386
BEGIN DESCRIPTION:
Buck Creek 59427.6
END DESCRIPTION:
XS GIS Cut Line= 3
      1628216.08      6844580.14      1628867.09      6844875.27
      1629335.87      6845331.03
#Sta/Elev= 30
  4285.4 1843.47  4342.7 1834.76  4405.8  1833.8  4458.1 1834.06  4486.7 1832.58
  4503.8  1833.5  4532.9 1832.15  4538.4 1831.06  4561.5 1830.78  4659.3 1831.03
  4676.9 1831.61  4682.4 1832.96  4780.3 1834.29  5002.2 1831.37  5021.9 1829.63
  5022.4 1829.13  5035.8 1829.63  5078.5 1830.21  5156.2 1833.74  5255.2  1834.9
  5283.5 1832.75  5304.6 1834.26  5311.8 1833.66  5318.8  1834.7  5368.4 1835.69
  5446.1  1834.8  5460.2 1835.69  5488.5 1841.17  5559.3 1849.07    5654 1854.15
#Mann= 4 ,-1 , 0
  4285.4     .12       0  4405.8     .05       0  5021.9     .05       0
  5035.8     .05       0
Bank Sta=5021.9,5035.8
XS Rating Curve= 0 ,0
Exp/Cntr=0.3,0.1

Type RM Length L Ch R = 1 ,59042   ,345,345,345
BEGIN DESCRIPTION:
Buck Creek 59041.59
END DESCRIPTION:
XS GIS Cut Line= 3
      1628044.63      6844619.21      1628530.72      6845016.33
      1629040.34      6845536.79
#Sta/Elev= 30
  4375.7 1846.14  4460.4    1842  4495.6 1834.89  4509.9 1833.38  4581.3 1832.15
  4595.7 1829.32    4609 1828.56  4687.3 1831.02  4929.9 1833.96  4979.5 1830.09
    4993 1827.74  4993.5 1827.24  5007.6 1827.74  5078.3 1830.93  5106.5 1830.55
  5113.7 1829.35  5191.4  1830.3  5219.7 1829.47  5226.8 1830.93  5233.8 1830.07
    5241 1831.44    5248  1830.1  5290.4  1832.9    5340 1832.78  5389.4 1834.17
    5439 1837.86  5537.9 1842.63  5601.6 1848.19  5672.3 1850.27  5731.8 1854.23
#Mann= 4 ,-1 , 0
  4375.7     .12       0  4581.3     .05       0    4993     .03       0
  5007.6     .05       0
Bank Sta=4993,5007.6
XS Rating Curve= 0 ,0
Exp/Cntr=0.3,0.1

Type RM Length L Ch R = 1 ,58697   ,562,562,562
BEGIN DESCRIPTION:
Buck Creek 58696.96
END DESCRIPTION:
XS GIS Cut Line= 3
       1627814.6      6844814.53      1628352.77       6845287.6
      1628806.33      6845721.62
#Sta/Elev= 30
  4280.6 1842.47  4347.5 1839.14  4403.5 1834.57  4439.6 1833.41  4509.8 1828.14
  4552.5 1828.62    4581 1829.81  4630.3 1829.16  4693.9 1831.05  4836.2 1831.68
  4956.7 1831.19  4977.6 1829.96  4985.2 1827.67  4991.8  1827.6  4995.3 1825.84
    5006 1825.67  5012.8 1824.01  5013.3 1823.51  5027.5 1824.01  5048.5 1826.29
  5062.7 1828.77  5083.7 1828.14  5140.3 1828.71  5175.9 1832.13  5218.3 1834.48
  5387.8 1840.03  5465.8 1846.41  5515.2 1847.57  5536.6 1849.34  5624.9 1852.76
#Mann= 3 ,-1 , 0
  4280.6     .05       0  5012.8     .03       0  5027.5     .05       0
Bank Sta=5012.8,5027.5
XS Rating Curve= 0 ,0
Exp/Cntr=0.3,0.1

Type RM Length L Ch R = 1 ,58135   ,90,90,90
BEGIN DESCRIPTION:
Buck Creek 58134.66
END DESCRIPTION:
XS GIS Cut Line= 5
      1627794.92      6844785.44      1628119.28       6845462.5
      1628131.91      6845727.67      1628164.46      6845782.36
      1628355.86      6846021.93
#Sta/Elev= 30
  3921.4 1844.45  4027.7 1838.71  4057.3  1835.5  4123.8 1831.45  4146.5 1830.18
  4179.3 1830.28  4208.9 1827.85  4356.7 1828.54  4441.1 1829.84  4599.7 1829.97
  4717.7  1829.5  4787.8 1828.04  4827.8 1830.63  4837.8 1830.62  4907.9 1822.64
  4927.9  1821.3  4935.3 1819.58  4953.9 1818.87  4954.4 1818.37  4968.6 1818.87
  4991.5 1819.73  5047.7 1819.66  5055.7 1823.16    5091 1831.11  5148.6 1836.28
  5204.6 1842.78  5226.1 1843.95  5247.9 1843.89  5254.3 1844.88  5307.9 1847.71
#Mann= 3 ,-1 , 0
  3921.4     .05       0  4953.9     .05       0  4968.6     .05       0
Bank Sta=4953.9,4968.6
XS Rating Curve= 0 ,0
Exp/Cntr=0.3,0.1

Type RM Length L Ch R = 1 ,58045   ,66,66,66
BEGIN DESCRIPTION:
Buck Creek 58045.29
END DESCRIPTION:
XS GIS Cut Line= 5
      1627750.68      6844832.38      1628068.09      6845447.04
      1628057.69      6845708.14      1628131.91      6845863.09
      1628261.08      6846037.47
#Sta/Elev= 30
  3876.6 1843.24    3973 1838.12  4025.6 1833.25    4142 1830.69  4180.7 1827.04
  4202.9 1827.97  4330.1 1828.24  4402.2 1829.59  4485.2  1829.1  4589.3 1829.89
  4609.4 1828.68  4649.4 1829.47  4699.4  1826.5  4719.5 1827.41  4729.5  1825.9
  4732.1 1824.72  4732.6 1824.22  4746.8 1824.72  4759.5 1829.41  4768.1 1829.84
  4773.1 1828.84  4799.5 1832.95  4832.4  1832.5  4857.7 1833.78    4903 1832.48
  4953.9 1832.41  5035.3 1833.33  5064.5  1831.8  5164.7 1843.83  5218.5 1844.29
#Mann= 3 ,-1 , 0
  3876.6     .05       0  4732.1     .03       0  4746.8     .05       0
Bank Sta=4732.1,4746.8
XS Rating Curve= 0 ,0
Exp/Cntr=0.3,0.1

Type RM Length L Ch R = 1 ,57979   ,173,173,173
BEGIN DESCRIPTION:
Buck Creek 57978.53
END DESCRIPTION:
XS GIS Cut Line= 6
      1627675.16      6844907.91      1628012.05      6845475.43
      1627986.08      6845734.18      1628034.25      6845857.88
      1628085.03      6845909.96      1628223.04      6846076.61
#Sta/Elev= 30
  3875.9 1840.46  3926.4 1838.75  4000.5 1833.09  4160.3  1830.5  4212.9 1828.76
  4240.2 1826.95  4314.2 1826.75  4341.5 1827.63  4548.5 1828.81    4639 1826.71
    4649 1826.22  4655.3  1824.3  4660.3 1825.63  4689.2  1826.8  4719.4 1826.83
  4779.7  1825.8  4795.3 1824.69  4830.6 1825.29  4853.1 1822.55  4853.6 1822.05
  4867.8 1822.55  4914.8 1824.33  4936.4 1823.03  4971.6 1824.75    4993 1823.98
  5007.3 1825.14  5042.4 1830.92  5085.4 1834.63  5155.7 1843.15  5217.8 1844.37
#Mann= 3 ,-1 , 0
  3875.9     .05       0  4853.1     .03       0  4867.8     .05       0
Bank Sta=4853.1,4867.8
XS Rating Curve= 0 ,0
Exp/Cntr=0.3,0.1

Type RM Length L Ch R = 1 ,57806   ,403,403,403
BEGIN DESCRIPTION:
Mapping XS d56d5a14
END DESCRIPTION:
XS GIS Cut Line= 3
      1627732.43      6845493.79      1627854.84      6845842.78
      1628179.44      6846414.07
#Sta/Elev= 30
  4413.6 1830.14  4598.2 1828.92  4677.9    1829  4788.8 1827.75  4816.2 1826.69
  4891.1 1825.17  4904.4 1823.72  4950.3 1823.21  4954.6 1822.12  4955.1 1821.62
  4968.9 1821.62  4969.4 1822.12  4993.5 1824.25  4999.3  1826.7  5020.9 1829.46
    5031 1830.05  5042.5 1831.67  5074.2 1833.75  5101.6 1837.38  5123.2 1839.05
  5182.4 1841.34    5204 1841.41  5226.5 1843.43  5235.7 1843.24  5284.7 1845.24
  5294.8 1845.04  5300.6 1845.73  5316.5 1845.96  5322.2 1846.74  5440.5 1848.26
#Mann= 3 ,-1 , 0
  4413.6     .05       0  4954.6     .05       0  4969.4     .05       0
Bank Sta=4954.6,4969.4
XS Rating Curve= 0 ,0
Exp/Cntr=0.3,0.1

Type RM Length L Ch R = 1 ,57403   ,214,214,214
BEGIN DESCRIPTION:
Buck Creek 57403.22
END DESCRIPTION:
XS GIS Cut Line= 3
      1627694.41      6845711.56      1627677.05      6846317.51
      1627702.96      6846614.59
#Sta/Elev= 30
  4395.7    1828  4562.2 1826.71  4702.3  1826.7  4712.3 1826.95  4762.3 1826.23
  4792.3 1826.52  4802.3 1826.06  4822.3 1826.08  4832.3 1825.74  4852.3 1823.76
  4882.3    1822    4935 1820.71  4935.5 1820.21  4949.3 1820.21  4949.8 1820.71
  5004.7 1821.79  5022.5 1823.12  5031.7 1824.33  5036.7 1825.54  5042.5  1826.3
  5072.7 1827.45  5132.9 1830.88  5149.5 1831.34    5163 1832.42  5183.1 1832.59
  5193.1 1833.16  5203.1 1832.93  5253.3 1833.31  5267.2 1833.83  5300.1 1834.19
#Mann= 3 ,-1 , 0
  4395.7     .05       0    4935     .05       0  4949.8     .05       0
Bank Sta=4935,4949.8
XS Rating Curve= 0 ,0
Exp/Cntr=0.3,0.1

Type RM Length L Ch R = 1 ,57189   ,355,355,355
BEGIN DESCRIPTION:
Mapping XS 01dbdd1c
END DESCRIPTION:
XS GIS Cut Line= 4
      1626993.29      6845603.62      1627475.06      6846384.88
      1627613.95      6846610.57      1627691.02      6846644.82
#Sta/Elev= 30
  3985.7 1835.73  3997.6 1835.26  4003.5    1834  4018.9 1832.81  4302.7 1828.77
  4702.5 1826.05  4797.1 1825.17  4839.7 1823.79  4876.4 1823.82  4891.8 1824.28
  4897.6 1825.49    4913 1825.64  4928.5  1822.5  4934.3 1819.64  4942.5 1817.22
  4948.2 1814.19  4948.7 1813.69  4963.1 1814.19  4986.4    1815  4992.3 1817.74
  5023.1 1824.09  5050.3 1830.72  5059.8 1830.27  5065.7 1828.04  5081.1 1825.79
  5164.8  1830.8  5191.6  1831.4  5198.1 1832.38  5226.8 1832.35  5252.9  1834.2
#Mann= 3 ,-1 , 0
  3985.7     .05       0  4948.2     .03       0  4963.1     .05       0
Bank Sta=4948.2,4963.1
XS Rating Curve= 0 ,0
Exp/Cntr=0.3,0.1

Type RM Length L Ch R = 1 ,56834   ,431,431,431
BEGIN DESCRIPTION:
Buck Creek 56834.4
END DESCRIPTION:
XS GIS Cut Line= 3
      1626471.62      6846636.35      1627258.13       6846686.7
      1627721.68      6846660.75
#Sta/Elev= 30
  4212.9 1838.62  4319.3  1834.4  4466.8 1825.66  4472.7 1826.21    4547 1824.14
  4626.1 1823.75  4657.2 1821.82  4697.3 1820.74  4747.4 1822.13  4807.5 1822.63
  4847.6 1820.94  4907.7 1820.48    4948 1821.22    5001 1819.68  5020.5 1818.45
    5021 1817.95  5034.9 1817.95  5035.4 1818.45    5048 1819.44  5065.1  1822.4
  5070.1 1820.93    5088  1823.2    5098 1823.59  5188.2 1824.74  5249.7 1826.41
  5358.4 1831.18  5368.5 1830.94  5424.3 1834.23  5429.3 1833.98  5465.3 1835.41
#Mann= 3 ,-1 , 0
  4212.9     .05       0  5020.5     .05       0  5035.4     .05       0
Bank Sta=5020.5,5035.4
XS Rating Curve= 0 ,0
Exp/Cntr=0.3,0.1

Type RM Length L Ch R = 1 ,56403   ,420,420,420
BEGIN DESCRIPTION:
Buck Creek 56403.11
END DESCRIPTION:
XS GIS Cut Line= 3
      1626412.64      6846881.14      1626909.17      6846891.56
      1627709.51      6846868.99
#Sta/Elev= 30
  4503.7 1839.36  4546.1 1838.55  4586.1 1836.05  4606.1 1835.75  4626.1 1833.97
  4656.1 1833.41  4676.1 1832.07  4686.1 1830.65  4726.1 1828.49  4756.1 1825.33
  4846.1 1821.39  4876.1 1820.61  4906.2 1821.49  4956.2 1821.32  4966.2 1818.73
  4978.7 1816.74  4979.2 1816.24  4993.2 1816.24  4993.7 1816.74  5026.2 1818.62
  5076.2  1819.5  5096.2 1821.03  5196.3 1820.96  5276.3 1822.61  5426.3 1824.28
  5486.4 1824.31  5536.4 1826.06  5566.4 1825.56  5706.5 1831.73    5801 1835.02
#Mann= 3 ,-1 , 0
  4503.7     .05       0  4978.7     .05       0  4993.7     .05       0
Bank Sta=4978.7,4993.7
XS Rating Curve= 0 ,0
Exp/Cntr=0.3,0.1

Type RM Length L Ch R = 1 ,55983   ,478,478,478
BEGIN DESCRIPTION:
Buck Creek 55983.37
END DESCRIPTION:
XS GIS Cut Line= 3
      1626236.23      6847162.97      1626711.94      6847239.36
      1627819.59      6847558.81
#Sta/Elev= 30
  4521.2  1842.1  4560.5 1840.72  4580.1 1841.03  4621.2 1838.19  4641.5 1838.46
  4661.8 1836.75  4702.3 1836.06    4714 1836.72  4752.9 1833.57  4803.5 1832.54
  4884.6  1826.6  4925.1 1822.36  4955.5 1820.65  5011.5 1813.73    5012 1813.23
  5026.5 1813.73    5027 1814.51  5052.6 1815.58    5079  1819.5  5131.1 1821.14
  5415.2 1819.98  5733.7 1823.98  5777.8 1825.04  5797.2 1826.63  5806.2 1824.86
  5811.4 1824.84  5828.4 1826.03  5990.1 1830.26  6067.8 1834.04  6155.8 1836.03
#Mann= 3 ,-1 , 0
  4521.2     .05       0  5011.5     .05       0  5026.5     .05       0
Bank Sta=5011.5,5026.5
XS Rating Curve= 0 ,0
Exp/Cntr=0.3,0.1

Type RM Length L Ch R = 1 ,55505   ,135,135,135
BEGIN DESCRIPTION:
Buck Creek 55505.01
END DESCRIPTION:
XS GIS Cut Line= 4
      1626378.72      6847697.87      1626755.43      6847701.34
      1627021.06      6847727.38      1627541.81      6847791.39
#Sta/Elev= 30
  4623.7 1830.35    4640  1829.2    4780 1826.15    4900 1821.59    4930 1819.55
    4940 1818.39    4970 1809.69  4990.2 1807.77  4990.7 1807.27  5004.8 1807.27
  5005.3 1807.77    5010 1808.31  5016.3  1811.4  5021.3 1810.99  5030.1 1812.59
  5040.2 1813.01  5060.3 1815.21  5080.4 1813.83  5122.8 1818.33  5219.2 1817.49
  5224.3 1817.03  5301.5 1817.19  5382.1  1819.3  5563.9 1821.65  5613.9 1823.05
    5634 1824.14  5645.2 1824.05  5664.2 1825.39  5674.3 1825.29    5792 1830.08
#Mann= 3 ,-1 , 0
  4623.7     .05       0  4990.2     .05       0  5005.3     .05       0
Bank Sta=4990.2,5005.3
XS Rating Curve= 0 ,0
Exp/Cntr=0.3,0.1

Type RM Length L Ch R = 1 ,55370   ,109,109,109
BEGIN DESCRIPTION:
Buck Creek 55369.73
END DESCRIPTION:
XS GIS Cut Line= 3
      1626328.37      6847796.83      1626807.52      6847805.51
      1627439.49      6847951.35
#Sta/Elev= 30
  4523.2 1830.37  4649.8 1827.12  4659.8 1827.29  4669.8 1828.86  4679.9 1828.54
  4699.9 1825.38  4749.9 1824.48  4759.9 1823.24  4829.9 1821.51  4859.5 1821.74
  4864.5 1819.71  4869.9 1819.31  4979.9 1821.99  4989.9 1819.06  4998.7 1813.13
  5012.8 1812.09  5013.3 1811.59  5027.9 1812.09  5030.6 1812.61  5051.2 1821.83
  5071.7 1820.92  5078.5 1819.47  5083.6 1820.16  5092.2 1819.72  5121.3 1816.44
  5174.3 1815.88  5225.6  1817.2  5441.1 1817.72    5513 1821.49    5651 1824.98
#Mann= 3 ,-1 , 0
  4523.2     .05       0  5012.8     .05       0  5027.9     .05       0
Bank Sta=5012.8,5027.9
XS Rating Curve= 0 ,0
Exp/Cntr=0.3,0.1

Type RM Length L Ch R = 1 ,55261   ,308,308,308
BEGIN DESCRIPTION:
Buck Creek 55261.09
END DESCRIPTION:
XS GIS Cut Line= 4
      1626366.08       6847864.1      1626851.79      6847899.26
      1626975.49      6847922.69      1627440.78      6848091.65
#Sta/Elev= 30
  4512.9 1829.98  4531.9 1828.87  4682.3 1824.29  4802.6 1819.71  4842.7 1817.23
  4902.8 1815.29  4910.5 1814.37  4915.6 1814.92  4922.9  1814.3    4953 1815.05
    4973 1812.38  4983.1  1812.6    4999 1814.13  5033.7 1814.18  5056.6 1811.96
  5057.1 1811.46  5071.4 1811.46  5071.9 1811.96  5076.6 1813.96  5125.8 1815.61
  5128.6 1816.76  5146.5 1817.54  5263.6 1816.53  5276.3 1815.79  5348.7 1815.58
  5393.5  1816.2  5418.7 1817.63    5480 1819.25  5535.9 1823.26  5620.8 1826.03
#Mann= 3 ,-1 , 0
  4512.9     .05       0  5056.6     .05       0  5071.9     .05       0
Bank Sta=5056.6,5071.9
XS Rating Curve= 0 ,0
Exp/Cntr=0.3,0.1

Type RM Length L Ch R = 1 ,54953   ,320,320,320
BEGIN DESCRIPTION:
Buck Creek 54953.07
END DESCRIPTION:
XS GIS Cut Line= 3
      1626318.79      6848184.33       1627003.7      6848155.68
      1627501.84      6848236.11
#Sta/Elev= 30
  4313.5 1832.46    4345 1830.32  4389.8 1828.83  4409.8    1827  4469.8  1823.7
  4489.9  1821.8  4529.9  1819.4  4539.9 1819.42  4569.9 1817.81    4600 1816.99
  4819.5  1816.2  4870.2 1813.98  4920.2 1814.32  4950.3 1812.38  4972.6 1809.34
  4973.1 1808.84  4987.4 1808.84  4987.9 1809.34  4997.2 1811.04  5002.2 1811.04
  5020.6 1814.52  5040.4  1816.3  5101.6 1815.43    5132 1813.92  5162.4 1813.79
  5223.2 1816.56  5297.5 1821.67  5415.6  1827.1    5421 1827.85  5503.6 1830.62
#Mann= 3 ,-1 , 0
  4313.5     .05       0  4972.6     .05       0  4987.9     .05       0
Bank Sta=4972.6,4987.9
XS Rating Curve= 0 ,0
Exp/Cntr=0.3,0.1

Type RM Length L Ch R = 1 ,54633   ,323,323,323
BEGIN DESCRIPTION:
Buck Creek 54632.66
END DESCRIPTION:
XS GIS Cut Line= 3
      1626294.23      6848412.71      1627058.17      6848461.32
      1627581.24      6848468.25
#Sta/Elev= 30
  4237.6 1830.75  4258.4 1829.55  4298.5 1828.48  4358.6 1823.46  4378.6 1821.39
  4478.9 1814.95  4599.1 1814.13  4639.2 1814.57  4719.5 1814.35  4819.5 1814.93
  4879.7 1813.03  4909.7 1813.96  4929.8 1813.64  4939.8 1812.89  4969.8 1811.83
  5003.1 1811.95  5009.9 1809.23  5012.3 1808.82  5012.8 1808.32  5027.1 1808.32
  5027.6 1808.82  5039.9 1812.01  5069.9  1815.3  5079.9 1816.01  5149.9 1817.81
  5189.9 1819.86  5229.9 1822.51  5379.9 1829.11  5429.9 1830.78  5526.2 1832.81
#Mann= 3 ,-1 , 0
  4237.6     .05       0  5012.3     .03       0  5027.6     .05       0
Bank Sta=5012.3,5027.6
XS Rating Curve= 0 ,0
Exp/Cntr=0.3,0.1

Type RM Length L Ch R = 1 ,54310   ,300,300,300
BEGIN DESCRIPTION:
Buck Creek 54310.15
END DESCRIPTION:
XS GIS Cut Line= 3
      1626236.99      6848607.15      1627003.05      6848767.75
      1627486.98      6848832.85
#Sta/Elev= 30
  4214.7  1827.2  4222.9 1827.37  4245.8 1826.03  4284.2 1824.92  4345.6 1820.17
  4406.8 1817.51  4427.2 1816.39  4435.2 1815.16  4447.7 1814.39  4490.3 1812.65
  4540.2 1812.15  4611.1 1813.15  4692.9 1811.49  4829.4 1813.81  4917.7 1812.55
  4929.3 1811.86  4948.3 1812.64  4968.8 1810.69  4989.2 1810.81  5033.2 1809.87
  5033.7 1809.37    5048 1809.37  5048.5 1809.87    5070 1812.67  5080.1 1812.95
  5120.5 1816.19  5150.7  1817.6  5201.2 1819.25  5337.1  1822.2  5485.7  1827.1
#Mann= 3 ,-1 , 0
  4214.7     .05       0  5033.2     .05       0  5048.5     .05       0
Bank Sta=5033.2,5048.5
XS Rating Curve= 0 ,0
Exp/Cntr=0.3,0.1

Type RM Length L Ch R = 1 ,54010   ,429,429,429
BEGIN DESCRIPTION:
Buck Creek 54009.58
END DESCRIPTION:
XS GIS Cut Line= 3
       1626229.6      6848763.83      1626984.82      6849062.45
      1627300.35      6849143.93
#Sta/Elev= 30
    4191 1820.76  4229.1 1818.66  4268.5 1817.77  4346.9 1814.72  4390.4 1812.14
  4465.9 1810.47  4544.3 1810.32  4583.9 1811.66  4622.7 1812.11  4809.3 1811.77
  4831.3 1812.45  4863.4 1809.97  4874.3  1807.5    4885 1807.73  4893.1 1808.77
  4898.5 1807.12  4917.3 1809.13  4928.2 1808.81  4947.2 1809.71  4999.2 1806.94
  4999.7 1806.44  5014.1 1806.44  5014.6 1806.94  5047.5 1813.78    5083 1816.75
  5123.7 1816.74  5220.2  1818.9  5245.6 1818.82  5292.5 1820.16    5329 1820.41
#Mann= 3 ,-1 , 0
    4191     .05       0  4999.2     .05       0  5014.6     .05       0
Bank Sta=4999.2,5014.6
XS Rating Curve= 0 ,0
Exp/Cntr=0.3,0.1

Type RM Length L Ch R = 1 ,53581   ,132,132,132
BEGIN DESCRIPTION:
Buck Creek 53581.01
END DESCRIPTION:
XS GIS Cut Line= 4
      1626061.51      6849121.55      1626521.54      6849258.25
      1626627.87      6849264.77      1626936.08      6849223.53
#Sta/Elev= 30
  4414.3 1822.65  4421.3 1822.74  4459.7 1820.87  4487.7  1818.7  4526.1 1817.04
  4559.3 1814.71  4564.5 1814.81  4647.5 1809.96  4678.7 1808.91  4735.3 1809.16
  4762.2 1811.07  4845.8 1811.43  4856.1 1809.29  4873.8 1803.61    4879 1803.44
  4893.4 1799.68  4959.6  1799.2  4960.1  1798.7  4974.5  1798.7    4975  1799.2
  5007.9 1800.73  5018.6 1802.49  5048.3 1804.01  5086.5 1807.38  5091.6 1805.66
  5108.8 1807.41    5129 1810.47  5139.1 1811.05  5219.8 1811.17  5311.7 1813.73
#Mann= 3 ,-1 , 0
  4414.3     .05       0  4959.6     .05       0    4975     .05       0
Bank Sta=4959.6,4975
XS Rating Curve= 0 ,0
Exp/Cntr=0.3,0.1

Type RM Length L Ch R = 1 ,53449   ,70,70,70
BEGIN DESCRIPTION:
Buck Creek 53449.09
END DESCRIPTION:
XS GIS Cut Line= 5
      1626054.94      6849195.32       1626517.2       6849327.7
      1626606.17       6849349.4      1626688.64      6849340.72
      1626910.03      6849264.75
#Sta/Elev= 30
  4519.4 1822.63  4546.4 1820.77  4571.5 1819.96  4592.3 1818.12  4685.9 1813.51
  4737.9 1810.02    4803 1808.22  4803.5 1807.72  4817.9 1807.72  4818.4 1808.22
  4871.1 1810.87  4935.5 1811.88  4943.8  1813.1    4949 1811.98  4956.3 1814.43
  4966.7 1816.07  4982.8 1815.29  5059.7  1815.8  5064.8 1816.39  5149.5 1816.19
  5154.5  1814.3  5181.5 1815.92  5197.9 1815.63  5203.2 1814.93  5223.8  1814.5
  5229.2 1812.92  5234.5 1813.13  5255.2 1810.05  5340.1 1810.63  5408.8    1813
#Mann= 3 ,-1 , 0
  4519.4     .05       0    4803     .05       0  4818.4     .05       0
Bank Sta=4803,4818.4
XS Rating Curve= 0 ,0
Exp/Cntr=0.3,0.1

Type RM Length L Ch R = 1 ,53379   ,395,395,395
BEGIN DESCRIPTION:
Buck Creek 53378.57
END DESCRIPTION:
XS GIS Cut Line= 4
      1626028.92      6849269.11      1626504.18      6849394.97
      1626695.15      6849410.16      1626947.45      6849272.15
#Sta/Elev= 30
  4507.6  1822.9  4555.3 1819.76  4669.1 1814.23  4676.6 1813.97  4681.8 1814.31
  4689.7 1813.19  4741.5 1810.04  4782.9 1808.41  4813.9 1808.59  4824.2 1809.13
  4832.3 1808.62  4855.3 1808.86  4886.3 1810.46    4938 1811.27  4958.7 1811.14
  4969.1 1810.03  4988.1 1804.88  5002.4 1804.22  5002.9 1803.72  5017.3 1803.72
  5017.8 1804.22  5040.2  1807.6  5110.4  1809.5  5228.6 1810.12  5250.4 1810.59
    5294 1809.88  5348.1 1809.91  5384.4 1810.89  5413.5 1812.29  5478.4 1813.56
#Mann= 3 ,-1 , 0
  4507.6     .05       0  5002.4     .05       0  5017.8     .05       0
Bank Sta=5002.4,5017.8
XS Rating Curve= 0 ,0
Exp/Cntr=0.3,0.1

Type RM Length L Ch R = 1 ,52984   ,170,170,170
BEGIN DESCRIPTION:
Buck Creek 52984.06
END DESCRIPTION:
XS GIS Cut Line= 6
      1625947.12      6849865.24      1626474.44      6849819.67
       1626634.6      6849719.41      1626660.64      6849682.95
      1626707.52      6849521.49      1627055.19       6849225.9
#Sta/Elev= 30
  4235.3  1818.4  4259.8 1817.36  4336.5 1816.07  4378.1 1815.14  4509.2 1809.46
  4624.6 1807.01  4654.7 1806.89  4755.1 1808.37  4968.3 1809.32  4976.9 1807.76
    4983 1807.74  4997.8  1800.8  5003.6  1799.9  5006.4 1797.08  5006.9 1796.58
  5021.3 1796.58  5021.8 1797.08  5029.1 1797.81  5055.7 1804.72    5061 1805.38
  5066.7 1807.59  5074.9 1808.09  5108.2 1808.95    5189 1809.11    5267  1810.1
    5323 1808.86  5330.7 1809.48  5365.8 1809.66  5443.8  1812.5  5622.9 1816.11
#Mann= 5 ,-1 , 0
  4235.3     .05       0  4336.5     .12       0  4509.2     .05       0
  5006.4     .05       0  5021.8     .05       0
Bank Sta=5006.4,5021.8
XS Rating Curve= 0 ,0
Exp/Cntr=0.3,0.1

Type RM Length L Ch R = 1 ,52814   ,386,386,386
BEGIN DESCRIPTION:
Buck Creek 52990.916
END DESCRIPTION:
XS GIS Cut Line= 4
      1625940.96      6849973.42      1626598.47      6849893.13
      1626809.09      6849743.25      1627162.25      6849175.65
#Sta/Elev= 30
  4079.1 1818.61  4123.5 1816.84  4197.1 1815.38  4364.4 1811.22  4445.8 1807.59
  4516.4 1805.81  4617.1 1807.33  4656.2 1806.94  4944.2 1808.87  4994.4  1805.3
  5029.7 1804.65  5065.1 1805.83  5080.1 1804.86  5095.4 1806.23  5101.3 1805.55
  5110.8 1805.89  5116.7 1804.32    5124 1804.98  5130.2  1804.3  5130.7  1803.8
  5145.1  1803.8  5145.6  1804.3  5153.3 1806.08  5168.6 1806.56  5182.8 1808.29
  5277.1 1809.93  5357.5 1812.36  5363.4 1813.34  5479.1 1815.73  5668.5 1817.79
#Mann= 5 ,-1 , 0
  4079.1     .05       0  4197.1     .12       0  4364.4     .05       0
  5130.2     .03       0  5145.6     .05       0
Bank Sta=5130.2,5145.6
XS Rating Curve= 0 ,0
Exp/Cntr=0.3,0.1

Type RM Length L Ch R = 1 ,52428   ,577,577,577
BEGIN DESCRIPTION:
Buck Creek 51987.43
END DESCRIPTION:
XS GIS Cut Line= 3
      1625787.04      6850099.79      1627055.55      6850028.73
      1627838.05       6850593.8
#Sta/Elev= 30
  3729.5 1822.99  3832.4  1819.9  3839.9 1819.67  4027.7 1814.12  4173.1 1811.11
  4390.4 1805.01  4548.7 1805.13  4799.1 1807.17  4909.3 1805.67  4939.4 1805.84
  4959.4 1807.14  4969.4 1805.87  4979.4 1803.27  4988.4 1797.34  4988.9 1796.84
  5006.1 1797.34  5012.6 1797.61  5021.1 1800.47  5027.3 1799.09  5035.8 1803.53
    5042 1803.13  5048.7 1805.55  5077.6  1806.2    5107  1808.9  5363.4 1813.66
  5440.3 1815.59  5536.3 1819.08  5801.1 1825.38  5829.6 1827.36  5965.2 1830.13
#Mann= 9 ,-1 , 0
  3729.5     .05       0  3832.4     .12       0  3839.9     .05       0
  4027.7     .12       0  4173.1     .05       0  4988.4     .05       0
  5006.1     .05       0  5363.4     .12       0  5440.3     .05       0
Bank Sta=4988.4,5006.1
XS Rating Curve= 0 ,0
Exp/Cntr=0.3,0.1

Type RM Length L Ch R = 1 ,51851   ,522,522,522
BEGIN DESCRIPTION:
Buck Creek 51850.89
END DESCRIPTION:
XS GIS Cut Line= 3
      1625797.45      6850386.25      1626703.73      6850381.04
      1627620.17      6850677.85
#Sta/Elev= 30
  4089.8 1821.84  4118.1 1820.84  4247.4 1819.39  4267.4  1817.9  4307.4 1817.14
  4467.4 1810.88  4637.4 1802.49    4654 1802.23  4697.4 1803.83  4897.4 1802.72
  4937.4 1805.18  4967.4 1805.07  4977.4 1804.38  4978.4 1800.41  4978.9 1799.91
  4996.3 1800.41  4999.3 1801.24  5018.5 1802.45    5050 1802.22  5081.5 1803.46
  5123.6 1803.81  5130.5 1803.56  5144.6  1800.9  5176.1  1802.4  5258.5  1803.9
  5354.5  1807.7  5459.9 1809.96  5594.8 1814.77  5818.2 1823.05  5959.4 1826.94
#Mann= 6 ,-1 , 0
  4089.8     .12       0  4118.1     .05       0  4978.4     .05       0
  4996.3     .05       0  5459.9     .12       0  5594.8     .05       0
Bank Sta=4978.4,4996.3
XS Rating Curve= 0 ,0
Exp/Cntr=0.3,0.1

Type RM Length L Ch R = 1 ,51329   ,699,699,699
BEGIN DESCRIPTION:
Buck Creek 51329.32
END DESCRIPTION:
XS GIS Cut Line= 3
      1625854.74      6850526.87       1626807.9       6850792.5
      1627860.02      6851261.27
#Sta/Elev= 30
  4016.6  1820.1  4172.6 1817.77  4374.8 1811.26  4432.1 1807.82  4463.3 1803.49
  4482.6 1798.68  4487.8 1798.51    4522 1801.74  4527.2  1801.4  4535.9 1802.35
  4577.4 1803.82  4608.6 1803.86  4961.5 1801.94  4992.7 1801.05  4997.1 1798.36
  4997.6 1797.86  5015.1 1798.36  5036.5 1799.69  5054.3  1803.1  5090.5 1804.82
  5243.8 1806.91  5349.5 1812.72  5378.2  1812.9  5523.1 1817.69  5841.6 1819.81
  5916.7    1819  5945.4 1819.49  5963.2 1820.67  6053.9 1821.72  6157.9 1824.34
#Mann= 3 ,-1 , 0
  4016.6     .05       0  4997.1     .05       0  5015.1     .05       0
Bank Sta=4997.1,5015.1
XS Rating Curve= 0 ,0
Exp/Cntr=0.3,0.1

Type RM Length L Ch R = 1 ,50630   ,434,434,434
BEGIN DESCRIPTION:
Buck Creek 50630.42
END DESCRIPTION:
XS GIS Cut Line= 3
      1625505.84      6850516.48       1626250.6      6850938.33
      1627401.64        6851605.
#Sta/Elev= 30
  4145.3 1823.69  4219.9 1822.39  4279.1 1821.25  4428.5 1819.27  4564.1 1817.92
  4682.4 1815.36  4879.9 1808.69  4952.2 1804.17  4960.3 1802.58  4968.1 1798.46
  4986.4 1794.45  4986.9 1793.95  5004.5 1794.45  5005.9 1796.99  5017.9 1798.86
    5041 1798.95  5064.1 1800.06    5172 1801.87  5318.3 1801.17  5391.5 1803.13
  5487.1 1804.29  5611.1 1805.67  5648.4    1807  5669.9  1806.5  5744.5  1808.2
  5862.8 1812.39  5883.6 1813.67  5985.5 1816.17    6152 1821.79  6331.4  1826.5
#Mann= 8 ,-1 , 0
  4145.3     .12       0  4219.9     .05       0  4279.1     .12       0
  4428.5     .05       0  4986.4     .05       0  5004.5     .05       0
  5487.1     .12       0  5862.8     .05       0
Bank Sta=4986.4,5004.5
XS Rating Curve= 0 ,0
Exp/Cntr=0.3,0.1

Type RM Length L Ch R = 1 ,50196   ,621,621,621
BEGIN DESCRIPTION:
Buck Creek 50195.99
END DESCRIPTION:
XS GIS Cut Line= 3
      1625420.67      6850897.73      1626155.01      6851345.63
      1627091.27        6851949.
#Sta/Elev= 30
  4148.1  1817.7  4179.9 1815.94  4332.9 1811.44  4501.3 1809.13  4929.3 1799.59
  4973.1 1794.61  4987.3 1794.16  4987.5 1792.86    4988 1792.36  5005.6 1792.86
    5024 1793.93  5045.1 1798.21  5054.3 1798.81  5135.8 1799.12  5162.9 1799.99
  5169.2  1801.6  5190.3 1800.58  5241.8 1801.55  5356.7 1801.54  5429.3 1803.01
  5436.5 1804.18  5459.6 1803.23  5607.7 1806.77  5733.9 1811.47  5819.4  1816.6
  5913.2 1820.02  6079.5 1822.34  6088.7 1823.08  6094.7 1822.44  6122.1 1822.78
#Mann= 5 ,-1 , 0
  4148.1     .05       0  4987.5     .05       0  5005.6     .05       0
  5135.8     .12       0  5607.7     .05       0
Bank Sta=4987.5,5005.6
XS Rating Curve= 0 ,0
Exp/Cntr=0.3,0.1

Type RM Length L Ch R = 1 ,49575   ,863,863,863
BEGIN DESCRIPTION:
Buck Creek 49574.71
END DESCRIPTION:
XS GIS Cut Line= 3
      1625056.06      6851158.13       1626024.8      6851923.75
      1627207.06      6852231.03
#Sta/Elev= 30
  3769.3 1813.83    4044 1804.83    4138 1802.22  4207.5 1801.33  4274.3 1801.03
  4295.1 1800.05  4708.7 1799.21  4800.4 1798.06    4893 1794.82  4921.8 1796.23
  4957.1 1794.33  5000.4 1794.74  5014.6 1794.29  5015.9 1793.39  5016.4 1792.89
    5034 1793.39  5035.3 1794.48  5045.8 1794.84  5081.2 1794.31  5121.7 1797.96
  5148.9 1798.55  5157.1 1800.13  5169.6 1801.03  5303.9 1805.12  5510.5 1812.86
    5522 1813.92  5644.9 1817.73  5714.3 1818.56  5800.6 1817.69  6225.6 1818.96
#Mann= 5 ,-1 , 0
  3769.3     .05       0    4044     .12       0  4207.5     .05       0
  5015.9     .05       0    5034     .05       0
Bank Sta=5015.9,5034
XS Rating Curve= 0 ,0
Exp/Cntr=0.3,0.1

Type RM Length L Ch R = 1 ,48712   ,607,607,607
BEGIN DESCRIPTION:
Buck Creek 48711.51
END DESCRIPTION:
XS GIS Cut Line= 3
      1624700.03      6851423.31      1625262.54      6852131.65
      1626240.83      6852506.31
#Sta/Elev= 30
  4098.4 1808.96  4197.5 1806.92  4283.2 1803.26  4418.6 1799.09  4468.3 1798.37
  4596.4 1794.89  4753.4 1794.45  4848.9 1795.17  4902.4 1795.18  4916.8 1793.53
  4931.3 1793.11  4937.7 1791.71  4945.7 1788.21    4960 1784.81  4971.9 1783.78
  4972.4 1783.28  4989.5 1783.28    4990 1783.78  5002.9 1786.62  5008.8 1789.64
  5016.3 1791.53  5032.9 1794.35  5038.8  1795.5  5063.5 1796.76  5112.6 1797.39
  5148.3 1798.79  5241.4 1799.37  5519.6 1801.62  5915.8 1808.05  6050.5 1808.46
#Mann= 6 ,-1 , 0
  4098.4     .05       0  4848.9     .12       0  4971.9     .05       0
    4990     .12       0  5032.9     .12       0  5241.4     .05       0
Bank Sta=4971.9,4990
XS Rating Curve= 0 ,0
Exp/Cntr=0.3,0.1

Type RM Length L Ch R = 1 ,48105   ,453,453,453
BEGIN DESCRIPTION:
Buck Creek 48105.32
END DESCRIPTION:
XS GIS Cut Line= 4
      1624002.15      6851834.79      1624856.29      6852449.36
      1625038.58      6852444.15      1625658.34      6852819.13
#Sta/Elev= 30
  3958.7 1807.42  4257.8 1803.39  4293.4 1801.48  4421.1 1799.08  4479.6  1796.5
  4492.3 1797.22  4586.7 1792.63  4836.9 1792.26  4880.1 1796.43  4909.6 1796.93
  4915.7 1793.84  4930.4 1795.74  4936.6 1792.07  4945.2 1792.13  4951.3 1789.14
  4956.9 1788.39  4957.4 1787.89  4975.1 1788.39  4980.8 1789.84  4995.5 1790.39
  5001.6 1788.96  5049.7  1791.2  5079.7 1790.98  5109.7  1793.7  5169.7 1793.05
  5214.4 1789.31  5245.4 1789.63  5478.2 1798.13  5726.5 1802.59  5917.7 1804.18
#Mann= 3 ,-1 , 0
  3958.7     .05       0  4956.9     .05       0  4975.1     .05       0
Bank Sta=4956.9,4975.1
XS Rating Curve= 0 ,0
Exp/Cntr=0.3,0.1

Type RM Length L Ch R = 1 ,47652   ,750,750,750
BEGIN DESCRIPTION:
Buck Creek 47651.96
END DESCRIPTION:
XS GIS Cut Line= 4
      1623637.54      6852230.61      1624668.79      6852834.78
      1624866.71      6852897.28      1625767.74      6853407.68
#Sta/Elev= 30
  3812.4 1803.81  4429.9 1796.89  4590.2  1791.9  4648.9 1791.34  4655.5 1792.09
  4664.5 1789.74  4678.7 1789.29  4830.6 1790.94  4889.2 1788.67  4898.9 1789.53
  4904.9 1788.18  4969.4 1788.91  4996.4 1787.64  4996.9 1787.14  5015.3 1787.64
  5032.4 1790.64  5037.6 1789.81  5045.6 1790.86  5064.7  1790.9    5070 1789.83
  5087.5 1789.23  5108.5 1791.17  5140.5  1792.4  5190.4 1793.46  5309.4 1794.71
  5546.1 1799.99  5661.4 1803.65  5787.8 1805.57  5983.2 1810.64  6250.7 1815.53
#Mann= 5 ,-1 , 0
  3812.4     .05       0  4996.4     .05       0  5015.3     .05       0
  5140.5     .12       0  5190.4     .05       0
Bank Sta=4996.4,5015.3
XS Rating Curve= 0 ,0
Exp/Cntr=0.3,0.1

Type RM Length L Ch R = 1 ,46902   ,818,818,818
BEGIN DESCRIPTION:
Buck Creek 46902.12
END DESCRIPTION:
XS GIS Cut Line= 3
       1623265.3       6852441.1      1624478.88        6853488.
      1625244.49      6853899.45
#Sta/Elev= 30
  3415.4 1801.23  3837.9 1797.88    4009 1795.17  4107.8 1794.39  4263.6 1788.04
  4412.8 1787.16  4490.7 1789.85    4498  1789.2  4597.1 1789.81    4845 1788.19
  4866.9 1788.81  4922.9 1787.08  4973.3 1786.59  4979.9 1786.08  4984.6 1784.31
  4985.1 1783.81  5003.2 1783.81  5003.7 1784.31  5008.4 1785.13    5046 1786.22
  5081.8 1791.35  5089.8 1791.82  5127.3  1793.2  5199.4 1797.52  5303.3 1801.15
  5407.2 1803.26  5494.8 1803.77  5649.5 1805.94  5797.1 1808.74  5887.3 1809.15
#Mann= 3 ,-1 , 0
  3415.4     .05       0  4984.6     .05       0  5003.7     .05       0
Bank Sta=4984.6,5003.7
XS Rating Curve= 0 ,0
Exp/Cntr=0.3,0.1

Type RM Length L Ch R = 1 ,46084   ,492,492,492
BEGIN DESCRIPTION:
Buck Creek 46084.35
END DESCRIPTION:
XS GIS Cut Line= 3
      1623046.61      6852493.25      1623780.96      6853842.17
      1624265.34      6854863.02
#Sta/Elev= 30
  3469.3 1800.56    3789 1798.14  3987.1 1797.84  4009.8 1796.94  4237.6 1793.43
  4312.3 1791.05  4377.8  1787.5  4431.1  1786.2  4791.9 1785.92  4835.6 1786.67
  4895.4 1784.24  4982.8 1783.23    4989  1782.1    5002 1781.48  5002.5 1780.98
  5021.2 1781.48  5021.7 1782.16  5033.8 1783.26  5055.9 1783.68  5072.7 1785.74
  5133.4 1785.97  5199.8 1789.34  5260.1  1790.2  5282.8 1791.38  5321.5 1791.46
  5515.7 1794.96  5543.9 1794.79  5589.4 1796.18  5808.6 1799.92  6135.1  1803.4
#Mann= 3 ,-1 , 0
  3469.3     .05       0    5002     .05       0  5021.2     .05       0
Bank Sta=5002,5021.2
XS Rating Curve= 0 ,0
Exp/Cntr=0.3,0.1

Type RM Length L Ch R = 1 ,45592   ,423,423,423
BEGIN DESCRIPTION:
Buck Creek 45592.21
END DESCRIPTION:
XS GIS Cut Line= 5
      1622923.68      6853854.53      1623385.96      6854012.96
      1623451.06        6854039.       1623535.7      6854041.17
      1623867.71      6854661.79
#Sta/Elev= 30
  4443.1 1792.75  4518.5 1792.48  4761.6 1787.35  4803.6 1787.48  4840.1 1785.41
  4902.7 1784.51    4934 1784.69  4958.2 1788.19  4982.5 1786.68  5065.9 1789.48
  5083.7 1788.79  5092.2 1789.35  5097.8 1788.55  5114.1 1783.01  5119.8 1782.58
  5126.4  1780.2  5126.9  1779.7  5145.7  1780.2    5158 1782.81  5196.2 1785.11
  5207.7 1787.86  5230.4 1787.04  5343.8 1790.45    5388  1792.1  5400.5 1793.38
  5623.7  1799.4  5629.3 1798.91  5705.8 1800.97  5755.3 1800.81  5790.4 1801.71
#Mann= 3 ,-1 , 0
  4443.1     .05       0  5126.4     .05       0  5145.7     .05       0
Bank Sta=5126.4,5145.7
XS Rating Curve= 0 ,0
Exp/Cntr=0.3,0.1

Type RM Length L Ch R = 1 ,45169   ,386,386,386
BEGIN DESCRIPTION:
Buck Creek 45169.15
END DESCRIPTION:
XS GIS Cut Line= 3
      1622739.98      6854211.32      1623198.28      6854349.33
      1623635.78        6854766.
#Sta/Elev= 30
  4524.2 1791.45  4550.3 1791.01  4654.8 1791.28  4759.2 1789.45  4832.3 1786.71
  4853.2 1785.22  4911.1 1782.57  4968.1 1781.44  4977.1 1779.93  4979.3 1778.31
  4979.8 1777.81  4998.2 1777.81  4998.7 1778.31  5013.6 1779.15  5041.9 1778.83
  5070.2 1779.28  5112.7 1782.16    5219 1787.16  5261.1 1787.88  5331.9  1790.4
  5339.1 1791.28    5346 1791.13  5360.2 1791.98  5388.5 1794.62  5409.9 1795.66
  5523.1 1797.21  5530.1 1797.89    5537 1799.41  5551.1 1800.54    5607 1802.27
#Mann= 3 ,-1 , 0
  4524.2     .05       0  4979.3     .05       0  4998.7     .05       0
Bank Sta=4979.3,4998.7
XS Rating Curve= 0 ,0
Exp/Cntr=0.3,0.1

Type RM Length L Ch R = 1 ,44783   ,662,662,662
BEGIN DESCRIPTION:
Buck Creek 44782.72
END DESCRIPTION:
XS GIS Cut Line= 3
      1622575.86      6854487.34      1623060.26      6854690.48
      1623435.28      6855029.04
#Sta/Elev= 30
  4474.9 1789.56  4528.2 1788.85  4549.9 1789.49  4734.2 1788.38  4802.3 1786.96
    4879 1783.77  4902.8 1782.05  4918.6 1779.87  4940.2 1777.96    4946 1775.63
  4946.5 1775.13  4964.9 1775.13  4965.4 1775.63  4972.8 1777.07    5037 1776.11
  5079.6 1777.39  5087.1 1778.73  5093.8 1778.81  5100.9 1781.26    5108 1781.58
  5214.1 1782.69  5263.4 1784.42  5277.6 1785.69  5334.4 1788.71  5356.1 1791.27
    5377 1791.59  5391.2 1793.09  5426.4 1794.98  5433.8 1795.88  5505.4 1798.25
#Mann= 3 ,-1 , 0
  4474.9     .05       0    4946     .05       0  4965.4     .05       0
Bank Sta=4946,4965.4
XS Rating Curve= 0 ,0
Exp/Cntr=0.3,0.1
