HEC-RAS study Buttonwillow Creek.prj: Buttonwillow Creek Base Level Engineering

--- Buttonwillow Creek.g01 (geometry) --- (continued)

Type RM Length L Ch R = 1 ,46809   ,347,347,347
BEGIN DESCRIPTION:
Mapping XS 7a5ab660
END DESCRIPTION:
XS GIS Cut Line= 4
        1575518.      6808437.96      1575778.39      6808414.53
      1576335.68      6808331.19      1576655.98      6808187.97
#Sta/Elev= 30
  4427.4 1850.49  4675.4 1848.86  4725.9 1847.76  4746.1 1847.78  4806.8 1845.53
  4887.6 1843.92  4897.4 1843.91  4907.9 1844.57  4971.6 1844.98  4978.6 1843.28
  4995.7 1842.85  4996.2 1842.35  5001.5 1842.35    5002 1842.85  5040.8 1845.06
  5160.6 1845.33  5293.4 1846.66  5368.5 1849.21  5397.2 1850.85  5414.9 1847.82
  5459.7 1848.19  5481.6 1848.91  5503.5 1852.08  5558.3 1852.38  5565.1  1854.5
  5570.6 1853.57  5588.3 1857.35  5593.8 1855.97  5599.9 1858.44  5603.2 1858.44
#Mann= 3 ,-1 , 0
  4427.4     .05       0  4995.7     .05       0    5002     .05       0
Bank Sta=4995.7,5002
XS Rating Curve= 0 ,0
Exp/Cntr=0.3,0.1

Type RM Length L Ch R = 1 ,46462   ,216,216,216
BEGIN DESCRIPTION:
Mapping XS 93f5c210
END DESCRIPTION:
XS GIS Cut Line= 2
      1575695.03      6808760.89      1576781.78      6808246.12
#Sta/Elev= 30
  4636.8 1849.76  4887.3  1847.2  4932.8 1846.07  4955.5 1844.99  4978.3 1843.57
  4990.9 1841.53  4997.8 1841.22  4998.3 1840.72  5003.7 1840.72  5004.2 1841.22
  5006.5 1842.42  5057.6 1843.51    5234 1843.62  5330.5 1844.96  5367.1 1844.92
    5478 1847.15    5518 1847.36  5523.5 1848.43    5533 1849.26  5555.2 1849.75
  5614.5  1853.5  5665.8 1856.03  5733.8 1858.01  5743.3 1857.65  5756.5 1858.56
  5765.4 1858.65  5773.7  1857.9  5779.3 1858.16  5787.5 1857.61  5839.3 1858.25
#Mann= 3 ,-1 , 0
  4636.8     .05       0  4997.8     .05       0  5004.2     .05       0
Bank Sta=4997.8,5004.2
XS Rating Curve= 0 ,0
Exp/Cntr=0.3,0.1

Type RM Length L Ch R = 1 ,46246   ,86,86,86
BEGIN DESCRIPTION:
Mapping XS f688bc11
END DESCRIPTION:
XS GIS Cut Line= 6
      1575689.84      6808815.57      1576116.93      6808755.67
      1576215.89      6808760.88      1576301.82      6808745.26
      1576325.26      6808693.17      1576890.31      6808273.28
#Sta/Elev= 30
  4510.4 1849.83  4748.9 1848.25  4929.6 1843.98  4941.7 1844.29  4949.7  1846.6
  4959.8 1846.78  5029.9 1837.44  5080.1 1835.61  5085.2 1834.32  5097.6 1834.22
  5098.1 1833.72  5103.5 1833.72    5104 1834.22  5121.2 1834.34  5127.2 1834.87
  5136.1 1834.35  5150.3  1835.8  5179.8 1841.31  5185.2 1841.31  5196.7 1843.42
  5202.9 1842.07  5217.5 1842.93    5253 1842.77  5432.4 1845.42  5503.3 1848.04
  5624.3 1854.01  5653.5 1854.16    5689 1855.62  5718.2 1855.31  5889.2 1857.97
#Mann= 3 ,-1 , 0
  4510.4     .05       0  5097.6     .05       0    5104     .05       0
Bank Sta=5097.6,5104
XS Rating Curve= 0 ,0
Exp/Cntr=0.3,0.1

Type RM Length L Ch R = 1 ,46160   ,107,107,107
BEGIN DESCRIPTION:
Mapping XS b49078f2
END DESCRIPTION:
XS GIS Cut Line= 6
      1575710.65      6808859.84      1576153.39      6808807.76
       1576226.3      6808846.82      1576327.87       6808833.8
      1576369.53      6808724.42      1576871.06      6808360.62
#Sta/Elev= 30
  4496.2 1849.77    4712 1848.66  4923.5 1843.69  4945.7 1844.62  4951.3 1846.28
  5017.1 1845.93  5043.6 1847.12  5104.1 1846.14  5123.1 1844.94    5136 1845.43
  5143.7 1843.99  5149.9 1845.48  5158.3 1843.89  5164.5  1845.5  5223.7 1844.45
  5243.7 1844.82    5265  1846.5  5273.5 1843.76  5291.2 1842.54  5291.7 1842.04
  5297.6 1842.54  5409.6 1843.44  5480.7 1845.25  5602.1 1850.18    5667 1851.63
  5696.4 1854.43    5732 1854.81  5752.8 1856.48  5773.7 1855.36  5876.9 1856.55
#Mann= 3 ,-1 , 0
  4496.2     .05       0  5291.2     .05       0  5297.6     .05       0
Bank Sta=5291.2,5297.6
XS Rating Curve= 0 ,0
Exp/Cntr=0.3,0.1

Type RM Length L Ch R = 1 ,46053   ,776,776,776
BEGIN DESCRIPTION:
Mapping XS 9edd31ec
END DESCRIPTION:
XS GIS Cut Line= 4
      1575848.69      6809180.16      1576114.32      6808977.03
      1576559.64      6808807.76      1577064.86      6808453.58
#Sta/Elev= 30
  4526.8 1848.46  4761.3 1847.66    4900 1845.71  4936.8 1842.69  4947.5  1841.3
  4954.9 1839.31  4957.1 1839.22  4957.6 1838.72    4963 1838.72  4963.5 1839.22
    4985 1841.43  5094.8 1842.29  5279.2 1841.21    5342 1841.18  5392.5 1841.83
  5455.3 1843.37  5470.1 1844.64  5484.9 1844.17  5520.7 1845.58  5550.3 1845.61
  5577.3 1846.63  5657.5 1848.09  5686.1 1849.51  5714.2 1851.97  5764.7 1852.96
  5808.2 1855.03  5821.4 1854.87  5886.8 1857.55  5922.5 1856.71  5954.6 1857.11
#Mann= 3 ,-1 , 0
  4526.8     .05       0  4957.1     .05       0  4963.5     .05       0
Bank Sta=4957.1,4963.5
XS Rating Curve= 0 ,0
Exp/Cntr=0.3,0.1

Type RM Length L Ch R = 1 ,45277   ,277,277,277
BEGIN DESCRIPTION:
Mapping XS b91af0a6
END DESCRIPTION:
XS GIS Cut Line= 3
      1575986.71      6809253.07      1576611.72      6809112.44
      1577085.66      6808734.85
#Sta/Elev= 30
  4132.9 1847.51  4418.1 1845.51  4544.7 1843.46  4612.9    1843  4715.4 1841.03
  4746.1 1841.58  4773.5 1843.54  4786.4 1843.91  4792.8 1843.34  4800.8 1843.56
  4807.2 1842.76    4836 1842.06  4842.4 1841.08  4856.9 1840.32    4985 1839.99
  5007.4  1838.2  5017.4 1837.95  5017.9 1837.45  5023.4 1837.45  5023.9 1837.95
  5034.6 1840.07  5057.1 1841.97  5113.1 1844.06  5199.6 1848.27  5220.4 1850.58
  5298.9 1851.29  5313.3 1851.76  5319.7 1853.09  5334.1 1854.07  5379.5 1855.05
#Mann= 3 ,-1 , 0
  4132.9     .05       0  5017.4     .05       0  5023.9     .05       0
Bank Sta=5017.4,5023.9
XS Rating Curve= 0 ,0
Exp/Cntr=0.3,0.1

Type RM Length L Ch R = 1 ,45000   ,125,125,125
BEGIN DESCRIPTION:
Mapping XS 902eb1c3
END DESCRIPTION:
XS GIS Cut Line= 6
      1576127.35      6809297.34      1576687.24       6809208.8
      1576794.01      6809245.26      1576937.24      6809195.78
      1576965.89      6809049.94      1577124.72      6808745.29
#Sta/Elev= 30
    4254 1846.96  4575.6 1843.87    4768 1840.71  4788.2 1842.51  4793.6 1845.14
  4798.7 1845.89  4833.9 1845.86  4865.4 1844.55  4891.5 1839.67  4896.7 1840.27
  4913.6 1836.24  4922.8  1834.9  4928.1 1835.34  4931.6 1833.35  4936.8 1833.35
  4940.3 1831.74  4973.8 1831.64  4974.3 1831.14  4980.3 1831.64    5065  1832.1
  5081.4 1834.88  5098.9 1834.85    5104 1835.92  5144.1 1837.25  5155.4  1838.9
    5195 1839.92    5315 1847.26  5457.5 1849.92    5518 1854.65  5577.4 1855.21
#Mann= 3 ,-1 , 0
    4254     .05       0  4973.8     .05       0  4980.3     .05       0
Bank Sta=4973.8,4980.3
XS Rating Curve= 0 ,0
Exp/Cntr=0.3,0.1

Type RM Length L Ch R = 1 ,44875   ,216,216,216
BEGIN DESCRIPTION:
Mapping XS 087cd54e
END DESCRIPTION:
XS GIS Cut Line= 6
       1576179.4      6809406.72      1576741.93      6809315.57
       1576911.2      6809315.57      1576986.72      6809253.07
      1577007.55      6809026.51      1577150.27      6808803.35
#Sta/Elev= 30
  4254.8 1846.14    4382 1845.55  4706.2 1842.49  4726.5 1841.66    4784 1840.87
  4784.5 1840.37    4790 1840.37  4790.5 1840.87  4797.4 1841.02  4823.7 1846.41
  4859.3 1846.47  4973.1 1844.94  5055.2 1845.64    5158 1844.49  5178.1  1843.6
  5198.2 1844.21  5231.5  1843.7  5248.4 1841.07  5258.4  1841.8  5268.4 1844.41
  5278.5  1844.8  5332.2 1845.76  5370.8 1847.71  5407.2 1848.69  5485.9 1849.53
  5552.7  1853.2  5558.6 1852.66  5573.8 1853.73    5589 1853.91    5595 1853.26
#Mann= 3 ,-1 , 0
  4254.8     .05       0    4784     .05       0  4790.5     .05       0
Bank Sta=4784,4790.5
XS Rating Curve= 0 ,0
Exp/Cntr=0.3,0.1

Type RM Length L Ch R = 1 ,44659   ,549,549,549
BEGIN DESCRIPTION:
Mapping XS 3912211c
END DESCRIPTION:
XS GIS Cut Line= 3
       1576471.1      6810055.14      1576945.05       6809646.3
      1577335.67      6808786.94
#Sta/Elev= 30
  4209.7 1845.73  4309.4 1845.76  4444.3 1844.09  4579.2 1843.46  4806.3 1840.31
  4835.6  1840.9  4946.7 1839.26  4964.2 1837.44  4969.7 1837.87  4976.6 1836.77
  4989.4 1836.77  4989.9 1836.27  4996.2 1836.77  5067.5 1838.37  5113.6 1837.92
  5136.7 1838.69  5196.2 1838.53    5229 1839.49  5257.5 1839.06  5303.7 1839.88
  5355.3 1839.43    5361 1841.52    5372 1841.45  5378.4 1840.42  5401.4 1841.71
  5545.3 1845.21    5597  1845.1  5666.2 1848.45  5746.3 1850.68  5779.6 1852.73
#Mann= 3 ,-1 , 0
  4209.7     .05       0  4989.4     .05       0  4996.2     .05       0
Bank Sta=4989.4,4996.2
XS Rating Curve= 0 ,0
Exp/Cntr=0.3,0.1

Type RM Length L Ch R = 1 ,44110   ,791,791,791
BEGIN DESCRIPTION:
Mapping XS 9adc6d4f
END DESCRIPTION:
XS GIS Cut Line= 3
      1577148.18      6810711.37      1577343.49      6809596.82
      1577557.05      6809057.71
#Sta/Elev= 30
  3661.2 1841.02  3684.9 1840.68  3776.3    1841  3979.3 1838.91  4060.6 1839.33
  4415.9 1839.04  4639.2 1837.31  4655.6 1837.96  4720.5 1837.32  4761.1 1837.81
  4769.3 1837.36  4814.4  1836.9  4868.4 1837.19  4976.5 1836.57  4995.5 1837.04
  5013.9 1835.77  5014.4 1835.27  5020.2 1835.27  5020.7 1835.77  5079.2  1837.5
  5084.6 1837.26  5108.9 1838.66  5133.3 1839.47  5192.7 1840.38  5232.5 1842.19
  5264.7 1842.67  5286.2 1844.34  5318.5 1844.62  5349.4 1846.55  5372.6 1846.81
#Mann= 3 ,-1 , 0
  3661.2     .05       0  5013.9     .05       0  5020.7     .05       0
Bank Sta=5013.9,5020.7
XS Rating Curve= 0 ,0
Exp/Cntr=0.3,0.1

Type RM Length L Ch R = 1 ,43319   ,624,624,624
BEGIN DESCRIPTION:
Mapping XS be3e711d
END DESCRIPTION:
XS GIS Cut Line= 3
       1577471.1      6810807.73      1577627.35      6809872.86
      1577876.95      6809202.03
#Sta/Elev= 30
  3958.7 1841.08  3968.6 1841.53  3978.7 1840.74  3988.8 1840.73  4012.7 1841.22
  4019.3 1840.29  4069.1 1839.45  4129.9 1839.05  4195.7  1837.6  4312.1 1836.43
  4769.5 1836.47  4910.3 1835.78  4945.9  1834.7    4971 1835.34  5004.3 1832.84
  5004.8 1832.34  5010.7 1832.34  5011.2 1832.84  5039.8 1834.05  5144.7 1834.76
  5197.7 1835.44    5228 1835.27  5288.7 1836.33  5295.8 1836.98  5319.1 1837.02
  5340.7 1837.96  5423.9 1841.02  5429.8 1841.65  5490.4 1842.06  5622.3  1844.1
#Mann= 5 ,-1 , 0
  3958.7     .05       0  5004.3     .05       0  5011.2     .05       0
  5144.7     .12       0  5340.7     .05       0
Bank Sta=5004.3,5011.2
XS Rating Curve= 0 ,0
Exp/Cntr=0.3,0.1

Type RM Length L Ch R = 1 ,42695   ,601,601,601
BEGIN DESCRIPTION:
Mapping XS f66287aa
END DESCRIPTION:
XS GIS Cut Line= 3
       1577593.5      6810773.88      1578171.62      6809948.38
      1578262.76       6809198.4
#Sta/Elev= 30
    3629 1841.68  3641.3 1841.96  3648.4 1840.33  3656.1 1840.01  3742.4 1839.09
    3793  1837.5  4215.8 1833.72  4266.4 1834.31  4453.9 1834.34  4717.8 1832.19
    4748 1830.85  4758.1  1832.4  4778.2 1830.94  4786.2 1831.85  4791.3  1831.1
  4801.8 1832.49  4808.4 1832.98    4873 1832.34  4989.8 1832.79  5006.4 1830.71
  5006.9 1830.21  5012.9 1830.21  5013.4 1830.71  5049.3 1833.14  5090.5 1835.46
  5118.2 1838.56  5123.3    1838    5200 1841.52  5231.5 1841.16  5392.3 1842.58
#Mann= 5 ,-1 , 0
    3629     .05       0  4801.8     .12       0  5006.4     .07       0
  5013.4     .12       0  5049.3     .05       0
Bank Sta=5006.4,5013.4
XS Rating Curve= 0 ,0
Exp/Cntr=0.3,0.1

Type RM Length L Ch R = 1 ,42094   ,370,370,370
BEGIN DESCRIPTION:
Mapping XS 4ab247f1
END DESCRIPTION:
XS GIS Cut Line= 4
        1577656.      6810786.91      1578512.76      6809953.59
      1578502.35      6809393.69      1578390.38       6809122.9
#Sta/Elev= 30
  3590.4 1842.05  3624.3  1842.4  3631.3 1841.14  3737.5 1839.08  3772.7 1837.31
  3808.2 1837.46  3857.6 1836.15  4041.5 1834.26  4140.5 1834.22  4225.4  1833.1
  4593.2 1832.92  4713.3 1831.29  4891.2 1831.72  4991.2  1829.9  4997.7 1828.28
  4998.2 1827.78  5004.2 1827.78  5004.7 1828.28  5011.2 1828.73  5021.2 1830.89
  5031.2 1831.34  5281.3 1834.21  5345.6 1835.38    5349 1836.11  5362.6 1836.69
  5384.2 1835.99  5407.7 1836.87  5470.8  1836.3  5492.4 1837.63  5638.6 1840.13
#Mann= 3 ,-1 , 0
  3590.4     .05       0  4997.7     .05       0  5004.7     .05       0
Bank Sta=4997.7,5004.7
XS Rating Curve= 0 ,0
Exp/Cntr=0.3,0.1

Type RM Length L Ch R = 1 ,41724   ,651,651,651
BEGIN DESCRIPTION:
Buttonwillow Creek 41302.081
END DESCRIPTION:
XS GIS Cut Line= 3
      1577708.11      6810846.78      1578805.09      6809827.92
      1579591.94      6809391.14
#Sta/Elev= 30
    3439  1843.3  3528.1 1843.21  3549.1 1842.65  3563.3 1841.11  3669.3 1837.37
    3896 1834.21    4002 1834.29  4171.7 1832.27  4688.6 1830.89  4752.1 1829.94
  4843.9 1830.44  4955.4 1828.96  4955.9 1828.46  4962.4 1828.96  5052.7 1829.97
  5112.2 1829.01    5134  1831.7  5187.7 1833.11    5222 1835.25  5236.9 1834.45
  5339.9 1836.44  5355.9 1838.26  5383.4 1837.49  5450.7  1839.4  5473.6 1838.78
  5599.4 1840.34  5664.9 1842.76  5679.5 1842.45  5686.6  1843.7  5836.1 1843.86
#Mann= 3 ,-1 , 0
    3439     .05       0  4955.4     .05       0  4962.4     .05       0
Bank Sta=4955.4,4962.4
XS Rating Curve= 0 ,0
Exp/Cntr=0.3,0.1

Type RM Length L Ch R = 1 ,41073   ,474,474,474
BEGIN DESCRIPTION:
Mapping XS e7d4de0b
END DESCRIPTION:
XS GIS Cut Line= 3
      1577942.47      6810961.38      1578325.26      6810464.01
      1579804.45      6810078.58
#Sta/Elev= 30
  3772.7 1843.81  3883.8  1842.6  3898.3 1841.12  3933.7 1840.88    3969 1838.62
  3991.5    1839  4047.8 1834.32  4758.9 1829.66  4792.7 1830.53  4915.7 1828.31
  4978.8 1828.62  5001.9  1826.9  5004.2 1825.25  5004.7 1824.75  5015.4 1825.25
  5037.2 1828.47  5071.8 1827.31  5082.9 1828.64  5115.9 1829.17  5320.7 1830.88
  5381.8 1832.68  5411.2 1832.13  5454.1 1833.07  5464.4 1833.74  5472.4 1835.66
  5495.4 1834.91  5536.8 1836.35  5553.4 1838.27  5593.9 1839.72  5928.9 1842.29
#Mann= 5 ,-1 , 0
  3772.7     .05       0  5004.2     .05       0  5015.4     .05       0
  5115.9     .12       0  5411.2     .05       0
Bank Sta=5004.2,5015.4
XS Rating Curve= 0 ,0
Exp/Cntr=0.3,0.1

Type RM Length L Ch R = 1 ,40599   ,986,986,986
BEGIN DESCRIPTION:
Mapping XS f4f44848
END DESCRIPTION:
XS GIS Cut Line= 3
      1578137.76      6811032.58      1578500.17      6810858.97
      1579690.79      6810431.74
#Sta/Elev= 30
    4168    1838  4262.7 1836.54  4284.3 1835.57  4468.9 1831.63    4620 1829.99
  4638.7 1830.56  4650.7 1829.29  4776.8 1829.27  4799.1 1827.88  4824.5  1829.1
    4850    1829  5029.1 1826.52  5106.2 1827.35  5121.3 1825.25  5171.8  1824.3
  5172.3  1823.8  5183.2  1824.3  5201.8 1828.27  5233.6 1827.69  5393.1 1830.87
  5412.8  1832.6  5424.9 1832.09  5456.8 1833.54  5467.4 1834.44  5474.3 1836.03
  5488.7 1835.22    5505  1836.3  5535.7 1836.48    5628 1840.53  5834.8 1842.74
#Mann= 5 ,-1 , 0
    4168     .05       0  4262.7     .12       0  4284.3     .05       0
  5171.8     .05       0  5183.2     .05       0
Bank Sta=5171.8,5183.2
XS Rating Curve= 0 ,0
Exp/Cntr=0.3,0.1

Type RM Length L Ch R = 1 ,39613   ,296,296,296
BEGIN DESCRIPTION:
Mapping XS 57d0cc53
END DESCRIPTION:
XS GIS Cut Line= 3
      1578361.29      6811410.18      1578951.56      6811347.25
      1579797.87      6810987.03
#Sta/Elev= 30
  4092.2 1840.51  4160.6 1838.09  4196.5 1834.48  4266.9 1830.99  4377.4 1828.14
  4404.7 1827.67  4598.8 1825.83  4627.8 1826.17  4632.8 1826.81  4690.4 1826.33
  4701.3 1827.08  4872.1  1824.9  4939.5 1825.17  4977.6 1823.72  4988.1 1821.88
  4988.6 1821.38  4999.2 1821.38  4999.7 1821.88  5001.2 1824.59  5053.9 1827.32
  5091.7 1827.22  5135.7 1829.01  5177.5 1829.38  5265.6 1832.36  5374.2 1833.72
  5406.5 1835.11  5435.6 1835.11  5517.4 1837.57  5548.1  1837.5  5605.6 1839.23
#Mann= 5 ,-1 , 0
  4092.2     .05       0  4377.4     .12       0  4404.7     .05       0
  4988.1     .05       0  4999.7     .05       0
Bank Sta=4988.1,4999.7
XS Rating Curve= 0 ,0
Exp/Cntr=0.3,0.1

Type RM Length L Ch R = 1 ,39317   ,445,445,445
BEGIN DESCRIPTION:
Mapping XS cb556a06
END DESCRIPTION:
XS GIS Cut Line= 2
       1578335.2       6811562.1      1580140.37      6811434.09
#Sta/Elev= 30
    4128 1840.59  4157.9 1840.31  4248.1 1836.46  4308.3 1833.15  4378.4 1830.95
  4388.5 1831.42  4400.7 1830.44  4488.7 1827.48  4528.8 1827.19    4619 1825.42
  4709.3  1824.9  4729.3 1825.55  4769.4 1825.64  4869.7 1825.31  4919.8 1824.27
  4949.9 1824.98  4959.2 1824.78  4969.9 1822.71  4979.9 1823.31  4994.2 1822.14
  4994.7 1821.64  5005.3 1821.64  5005.8 1822.14    5010 1824.08  5170.4 1825.38
  5300.7 1828.77  5310.8 1828.28  5451.1 1829.06  5771.9 1833.84  5937.7 1833.62
#Mann= 3 ,-1 , 0
    4128     .05       0  4994.2     .05       0  5005.8     .05       0
Bank Sta=4994.2,5005.8
XS Rating Curve= 0 ,0
Exp/Cntr=0.3,0.1

Type RM Length L Ch R = 1 ,38872   ,585,585,585
BEGIN DESCRIPTION:
Mapping XS 25484ac3
END DESCRIPTION:
XS GIS Cut Line= 3
      1578498.03       6811939.7      1579146.88       6811874.6
      1580409.88      6811783.45
#Sta/Elev= 30
  4040.6 1837.75    4118 1835.85  4168.2 1830.98  4205.6 1828.73    4319 1825.54
  4499.9 1823.28  4570.2  1824.3  4670.7 1823.67  4710.4 1824.76  4831.2 1822.64
    4855 1823.03  4861.3 1824.64  4871.3 1824.74  4931.5 1821.14  4961.5 1823.64
  4981.6 1824.11  5001.6  1822.3  5005.8 1820.88  5006.3 1820.38  5017.5 1820.88
  5051.8 1824.32  5101.9 1826.48  5172.1 1826.26  5302.4 1827.35  5432.8 1829.45
  5492.9 1828.78  5603.2 1829.77  5633.3 1828.46  5663.3 1831.03    5959  1833.6
#Mann= 3 ,-1 , 0
  4040.6     .05       0  5005.8     .05       0  5017.5     .05       0
Bank Sta=5005.8,5017.5
XS Rating Curve= 0 ,0
Exp/Cntr=0.3,0.1

Type RM Length L Ch R = 1 ,38287   ,530,530,530
BEGIN DESCRIPTION:
Mapping XS 68bf33f1
END DESCRIPTION:
XS GIS Cut Line= 3
      1578521.85      6812410.62       1579973.7      6812276.07
      1580399.07      6812074.24
#Sta/Elev= 30
  4112.8  1833.6  4307.8  1827.4  4467.5 1824.31    4598  1822.4  4718.5 1822.24
  4748.7 1822.83  4869.2 1822.34  4879.2  1821.7  4949.2 1820.95  4969.6 1820.16
  4989.7 1820.79  4999.7 1820.33  5003.7 1819.21  5004.2 1818.71  5015.4 1818.71
  5015.9 1819.21  5019.8 1820.92  5049.9 1822.73  5120.2 1823.84  5150.4 1823.31
  5200.6 1824.83  5220.7  1824.2  5240.8 1825.52  5461.7 1826.32  5511.9 1827.44
  5594.4 1827.21    5683 1828.42  5737.1 1827.42  6015.1  1831.1  6041.7 1830.28
#Mann= 3 ,-1 , 0
  4112.8     .05       0  5003.7     .05       0  5015.9     .05       0
Bank Sta=5003.7,5015.9
XS Rating Curve= 0 ,0
Exp/Cntr=0.3,0.1

Type RM Length L Ch R = 1 ,37757   ,565,565,565
BEGIN DESCRIPTION:
Mapping XS 1a5dbd9e
END DESCRIPTION:
XS GIS Cut Line= 4
       1578716.3      6813021.74       1579018.4      6812954.02
      1579843.06      6812533.88      1580344.76      6812440.14
#Sta/Elev= 30
  4320.7 1827.93  4498.3  1825.8  4565.3 1823.85    4705 1822.15  4943.6  1820.9
  4965.9 1819.95  4976.4 1818.12  4976.9 1817.62  4988.1 1817.62  4988.6 1818.12
  5010.4 1820.11  5115.9 1820.73    5154 1821.97  5182.6 1819.32  5221.3 1818.64
  5271.6 1819.94  5293.8 1822.32  5299.9 1822.35  5316.1 1820.47  5322.3 1822.12
  5332.7 1823.12  5367.2 1821.98  5382.8 1823.52  5488.4 1824.54  5524.3 1825.54
  5578.1 1825.41  5791.8 1827.83  5812.1 1826.83  5903.7 1828.77  6066.2 1830.25
#Mann= 3 ,-1 , 0
  4320.7     .05       0  4976.4     .05       0  4988.6     .05       0
Bank Sta=4976.4,4988.6
XS Rating Curve= 0 ,0
Exp/Cntr=0.3,0.1

Type RM Length L Ch R = 1 ,37192   ,174,174,174
BEGIN DESCRIPTION:
Mapping XS ce353894
END DESCRIPTION:
XS GIS Cut Line= 3
      1578797.57       6813272.6      1579649.13      6813236.14
      1580865.29      6813189.26
#Sta/Elev= 30
  4141.3 1828.08  4218.8 1825.84  4298.9 1825.35    4429 1822.83  4549.1 1822.36
  4609.2 1820.92  4649.2 1821.36  4899.4 1819.75  4929.4 1818.29  4959.5 1818.37
  4979.5 1817.05  5003.1 1816.95  5003.6 1816.45  5015.9 1816.95  5059.6 1819.26
  5139.6 1820.13  5159.6  1821.8  5179.6 1824.88  5209.7 1826.06  5239.7 1825.19
  5269.7 1825.93  5289.7 1821.61  5309.7 1821.11  5449.8 1823.02    5650    1823
  5854.6 1825.14  5880.2 1828.34  5920.2 1826.47  6080.3 1829.32  6210.7 1833.69
#Mann= 3 ,-1 , 0
  4141.3     .05       0  5003.1     .03       0  5015.9     .05       0
Bank Sta=5003.1,5015.9
XS Rating Curve= 0 ,0
Exp/Cntr=0.3,0.1

Type RM Length L Ch R = 1 ,37018   ,464,464,464
BEGIN DESCRIPTION:
Mapping XS b7a6df01
END DESCRIPTION:
XS GIS Cut Line= 2
      1579552.81      6813410.62      1580938.15       6813397.6
#Sta/Elev= 30
  4897.4 1822.62  4929.6 1822.25  4939.6 1821.19  4949.6 1819.37  4989.6 1818.65
  4999.6 1817.07  5013.2 1815.91  5013.7 1815.41  5025.5 1815.41    5026 1815.91
  5049.6 1816.48  5069.6 1818.33  5099.6 1817.55  5169.6 1818.55  5189.6 1817.72
  5209.6    1819  5349.6 1819.19  5399.6 1820.47  5519.6 1819.94  5629.6 1820.74
  5789.6 1823.52  5899.6 1824.41  5929.6 1825.41  5979.6 1825.13  6019.6 1826.24
  6099.6 1826.56  6149.6 1827.48  6189.6  1829.1  6229.6 1829.22  6282.8 1830.49
#Mann= 3 ,-1 , 0
  4897.4     .05       0  5013.2     .03       0    5026     .05       0
Bank Sta=5013.2,5026
XS Rating Curve= 0 ,0
Exp/Cntr=0.3,0.1

Type RM Length L Ch R = 1 ,36554   ,418,418,418
BEGIN DESCRIPTION:
Mapping XS efaeef73
END DESCRIPTION:
XS GIS Cut Line= 3
      1579557.98      6813871.56      1580362.67      6813798.64
      1580776.73      6813684.06
#Sta/Elev= 30
  4852.6 1821.03  4869.7 1821.08  4889.8 1819.86  4909.9 1816.91  4980.1 1816.19
  4983.8 1814.55  4984.3 1814.05  4996.1 1814.05  4996.6 1814.55  5010.3 1816.87
  5030.3 1817.49  5150.8 1818.35    5181 1817.75  5211.1 1818.36  5241.2 1818.38
  5251.2 1817.86  5371.7 1816.44  5401.9 1816.89  5421.9 1817.96    5442  1817.5
  5532.4 1817.71  5552.5 1817.89  5572.6 1820.08  5582.6 1820.55  5659.2 1822.85
  5685.3 1823.26  5963.9 1823.73  6014.9 1825.43  6036.5 1825.07  6090.2  1826.1
#Mann= 3 ,-1 , 0
  4852.6     .05       0  4983.8     .05       0  4996.6     .05       0
Bank Sta=4983.8,4996.6
XS Rating Curve= 0 ,0
Exp/Cntr=0.3,0.1

Type RM Length L Ch R = 1 ,36136   ,470,470,470
BEGIN DESCRIPTION:
Mapping XS e0124ce4
END DESCRIPTION:
XS GIS Cut Line= 3
      1579576.24      6814335.08      1580211.63       6813962.7
      1580700.65      6813848.25
#Sta/Elev= 30
  4761.1 1820.53  4817.6 1818.61  4861.1  1818.3  4898.3 1819.09  4919.8 1818.09
  4933.5 1818.46  4941.3 1817.97  4956.7 1818.03  4978.4 1816.18  4999.3  1812.2
  4999.8  1811.7  5011.7  1811.7  5012.2  1812.2  5014.7 1813.48  5037.1 1814.01
  5072.6 1816.36  5320.4 1817.39  5400.5 1816.35  5453.4 1816.35  5501.9 1816.81
  5521.6  1817.7  5543.7 1817.03  5562.6 1818.26    5581 1818.61  5586.2 1819.32
  5676.3 1821.87  5761.2 1822.35  5829.7 1823.38  5973.5 1823.42  5999.8 1823.91
#Mann= 3 ,-1 , 0
  4761.1     .05       0  4999.3     .05       0  5012.2     .05       0
Bank Sta=4999.3,5012.2
XS Rating Curve= 0 ,0
Exp/Cntr=0.3,0.1

Type RM Length L Ch R = 1 ,35666   ,377,377,377
BEGIN DESCRIPTION:
Mapping XS 24aa0504
END DESCRIPTION:
XS GIS Cut Line= 3
      1579576.18      6814512.18       1580003.3      6814488.74
      1580710.83      6814077.75
#Sta/Elev= 30
  4350.5 1820.96  4379.4 1818.87  4409.4 1817.99  4729.9 1816.39  4739.9    1816
  4749.9 1814.22  4753.4 1812.21  4753.9 1811.71  4765.9 1811.71  4766.4 1812.21
  4769.9 1815.12  4776.6 1816.33  4830.9  1815.5  4852.4 1814.34  4861.2 1815.44
  4883.9 1814.75  4964.2 1815.18    5013 1813.13  5050.3 1814.98  5146.3 1815.49
  5219.7 1817.13  5291.1 1817.46  5349.9 1818.48  5365.6 1819.52  5393.2    1819
  5430.2 1819.33  5483.2 1820.93  5504.7 1820.67  5569.3 1821.44  5596.5 1822.78
#Mann= 3 ,-1 , 0
  4350.5     .05       0  4753.4     .05       0  4766.4     .05       0
Bank Sta=4753.4,4766.4
XS Rating Curve= 0 ,0
Exp/Cntr=0.3,0.1

Type RM Length L Ch R = 1 ,35289   ,341,341,341
BEGIN DESCRIPTION:
Mapping XS a7b36c3d
END DESCRIPTION:
XS GIS Cut Line= 2
      1579557.97      6814694.47       1580899.1      6814733.54
#Sta/Elev= 30
  4252.6 1820.94  4279.6 1821.06  4299.7 1819.13  4329.7 1817.56  4479.7 1815.65
  4659.8 1815.18  4669.8 1812.32  4673.3 1811.96  4673.8 1811.46  4685.9 1811.46
  4686.4 1811.96  4689.8 1815.42  4779.9 1814.84  4799.9  1813.2  4809.9 1813.45
  4819.9 1812.79  4849.9 1814.01  4891.9 1813.68  4979.9 1814.77  4989.9 1814.14
    5020 1815.14    5080 1815.27    5150 1817.19    5210 1817.65  5260.1 1819.44
  5290.1 1819.33  5380.1 1821.27  5450.1 1821.64  5510.2 1823.28  5594.3 1823.83
#Mann= 3 ,-1 , 0
  4252.6     .05       0  4673.3     .05       0  4686.4     .05       0
Bank Sta=4673.3,4686.4
XS Rating Curve= 0 ,0
Exp/Cntr=0.3,0.1

Type RM Length L Ch R = 1 ,34948   ,450,450,450
BEGIN DESCRIPTION:
Mapping XS 19d4df84
END DESCRIPTION:
XS GIS Cut Line= 3
      1579537.15      6814853.33      1579883.51      6814926.24
      1580880.48       6815230.8
#Sta/Elev= 30
  4300.7 1820.82  4318.9 1820.43  4339.4 1820.95  4359.8 1820.48  4421.1 1816.81
  4445.7 1815.82  4490.4 1815.02  4745.7 1813.67  4760.8 1814.21  4802.6 1813.07
  4875.8 1813.81  4938.5 1813.39  4959.4 1812.75  4985.7 1813.16  5001.3 1812.71
  5005.2 1811.36  5005.7 1810.86  5017.8 1810.86  5018.3 1811.36  5018.5 1812.42
  5023.7 1812.74  5074.5 1814.56  5154.9 1815.77  5210.4 1815.85  5241.8 1816.92
    5433  1818.1  5471.8 1819.34  5536.6 1819.49  5607.7 1821.41  5697.1 1822.16
#Mann= 3 ,-1 , 0
  4300.7     .05       0  5005.2     .05       0  5018.3     .05       0
Bank Sta=5005.2,5018.3
XS Rating Curve= 0 ,0
Exp/Cntr=0.3,0.1

Type RM Length L Ch R = 1 ,34498   ,368,368,368
BEGIN DESCRIPTION:
Mapping XS f9231e7f
END DESCRIPTION:
XS GIS Cut Line= 3
      1579550.16      6814931.43      1580013.72      6815457.49
      1580810.34      6815439.27
#Sta/Elev= 30
  4531.2 1819.27  4539.7 1819.17  4546.4 1819.89    4589 1819.42  4617.5 1817.82
  4624.2  1816.5  4673.5 1814.93    4830 1812.98  4858.5 1813.07  4886.5 1812.26
  4928.7 1812.15  4964.7 1812.62  4985.6 1811.85  5006.5 1812.48  5034.9  1812.5
  5092.8 1811.75  5093.3 1811.25  5105.5 1811.25    5106 1811.75  5120.3 1812.28
  5323.7 1813.34  5423.7 1814.28  5428.8 1814.66  5433.8 1814.12  5533.7 1815.31
  5603.7 1817.34  5723.8 1818.92  5843.8 1821.85  5893.8 1821.44  6029.2 1822.28
#Mann= 3 ,-1 , 0
  4531.2     .05       0  5092.8     .05       0    5106     .05       0
Bank Sta=5092.8,5106
XS Rating Curve= 0 ,0
Exp/Cntr=0.3,0.1

Type RM Length L Ch R = 1 ,34130   ,573,573,573
BEGIN DESCRIPTION:
Mapping XS 5ae584bc
END DESCRIPTION:
XS GIS Cut Line= 3
      1579125.29      6815427.55      1579483.33      6815518.69
      1580370.45      6815807.17
#Sta/Elev= 30
  4450.4 1817.91  4501.7 1817.26  4522.3  1815.9  4550.8 1817.29  4596.9 1815.51
  4714.5 1815.42  4719.6 1814.06  4755.4 1814.65  4760.5 1813.24  4796.3 1813.82
  4867.5 1812.32  4874.2 1811.18  4894.2 1814.61  4916.2 1814.73  4931.4 1814.39
  4947.8 1811.99  4979.3 1811.53  5004.2  1809.9  5004.7  1809.4  5017.5  1809.9
    5116 1811.65  5410.5 1811.88  5536.7 1812.85  5568.2 1814.12  5612.7 1813.63
  5644.6 1814.51  5671.3 1816.71  5708.5 1816.31  5735.2 1818.24  5752.7 1818.43
#Mann= 3 ,-1 , 0
  4450.4     .05       0  5004.2     .03       0  5017.5     .05       0
Bank Sta=5004.2,5017.5
XS Rating Curve= 0 ,0
Exp/Cntr=0.3,0.1

Type RM Length L Ch R = 1 ,33557   ,510,510,510
BEGIN DESCRIPTION:
Mapping XS 6c71eb0e
END DESCRIPTION:
XS GIS Cut Line= 3
      1578767.15      6815707.47      1579292.36      6816033.02
      1580351.74      6816065.51
#Sta/Elev= 30
  4169.9 1817.66  4261.8 1815.93  4734.4  1810.7  4900.5 1810.31  4950.5 1811.45
  4970.5 1810.58  4980.6 1808.64  4983.9 1807.22  4984.4 1806.72  4996.8 1806.72
  4997.3 1807.22  5030.6 1810.33  5040.6 1811.97  5060.6 1812.88  5100.6 1811.16
  5114.5 1809.96  5120.6 1807.99  5130.6 1807.98  5160.6 1809.74  5190.6 1810.31
  5260.7 1810.89  5330.7  1810.3  5410.8 1811.16  5460.8 1810.85  5610.8 1812.18
  5670.9 1813.62  5720.9 1813.49  5765.8 1815.02  5770.9 1815.84  5847.7 1816.71
#Mann= 3 ,-1 , 0
  4169.9     .05       0  4983.9     .05       0  4997.3     .05       0
Bank Sta=4983.9,4997.3
XS Rating Curve= 0 ,0
Exp/Cntr=0.3,0.1

Type RM Length L Ch R = 1 ,33047   ,405,405,405
BEGIN DESCRIPTION:
Mapping XS 8ef426eb
END DESCRIPTION:
XS GIS Cut Line= 4
      1578669.54      6815944.05      1579238.11       6816317.3
      1579654.78      6816783.88      1580156.07      6816773.03
#Sta/Elev= 30
    4045 1816.65  4607.9 1809.16  4893.4 1809.55  4942.7 1808.07  4992.9 1808.05
  4999.6  1806.2  5000.3 1804.78  5000.8 1804.28  5013.8 1804.78    5021 1807.71
  5034.7 1809.16  5162.6 1807.54    5191 1809.02  5197.7 1811.08  5268.8 1810.09
  5289.7 1807.39  5303.9 1808.46  5311.4 1807.81  5318.1 1810.24  5325.6 1808.53
  5332.3  1809.4  5339.8  1807.1  5353.3 1807.07  5400.9 1808.98  5420.9 1808.32
    5551 1810.58    5571 1811.95    5691 1811.41    5821 1813.96  5852.1 1813.36
#Mann= 3 ,-1 , 0
    4045     .05       0  5000.3     .05       0  5013.8     .05       0
Bank Sta=5000.3,5013.8
XS Rating Curve= 0 ,0
Exp/Cntr=0.3,0.1

Type RM Length L Ch R = 1 ,32642   ,597,597,597
BEGIN DESCRIPTION:
Mapping XS 27a31130
END DESCRIPTION:
XS GIS Cut Line= 4
      1578393.07      6816544.45      1578920.83      6816721.53
       1579875.7      6816898.61      1580136.11      6816867.36
#Sta/Elev= 30
  4205.4 1815.41  4264.6 1814.32  4407.8 1813.46  4460.6 1812.19  4511.6 1812.01
  4555.5  1810.5  4597.7 1809.98  4611.5 1810.55  4643.1 1809.33  4737.7 1808.15
  4888.4 1807.98  4939.5 1806.34  4969.7 1806.84  4979.9 1806.46  4985.5 1803.07
    4986 1802.57  4999.1 1803.07  5000.2 1805.76  5010.4  1808.7  5051.1    1808
  5266.7 1808.01  5386.7  1806.8  5417.2 1808.46  5457.9 1806.75  5536.1 1807.27
    5594 1808.78  5722.3 1809.55  5742.6 1810.57  5883.6 1810.83  5995.5 1812.45
#Mann= 3 ,-1 , 0
  4205.4     .05       0  4985.5     .05       0  4999.1     .05       0
Bank Sta=4985.5,4999.1
XS Rating Curve= 0 ,0
Exp/Cntr=0.3,0.1

Type RM Length L Ch R = 1 ,32045   ,912,912,912
BEGIN DESCRIPTION:
Mapping XS 89f57541
END DESCRIPTION:
XS GIS Cut Line= 3
      1577858.31      6817044.44      1578643.06      6817148.61
      1579969.46      6816978.47
#Sta/Elev= 30
  4044.2 1823.35  4131.7 1818.19  4259.5 1814.37  4373.8 1812.66  4434.3 1809.49
  4706.7 1807.21  4792.8 1810.22    4858 1809.38  4898.3 1810.84  4948.7 1809.33
    4989 1804.56  5009.2 1804.18  5049.5 1806.12  5089.8 1802.91  5115.4 1806.85
  5281.4 1806.85  5311.6 1807.99  5321.7 1807.75  5341.9 1803.52  5362.1 1806.66
    5483 1807.18  5667.7 1805.85  5694.8  1805.3  5704.8  1804.5  5708.1 1802.79
  5708.6 1802.29  5721.7 1802.79    5725 1804.87  5765.3 1807.18  6173.1  1811.1
#Mann= 3 ,-1 , 0
  4044.2     .05       0  5708.1     .05       0  5721.7     .05       0
Bank Sta=5708.1,5721.7
XS Rating Curve= 0 ,0
Exp/Cntr=0.3,0.1

Type RM Length L Ch R = 1 ,31133   ,507,507,507
BEGIN DESCRIPTION:
Mapping XS c2be7645
END DESCRIPTION:
XS GIS Cut Line= 3
      1577837.53      6817381.25      1578577.08      6817471.53
      1579899.98      6817353.47
#Sta/Elev= 30
  3471.5 1818.88  3509.2  1818.7  3549.5 1816.83  3620.1 1815.97  3660.4 1814.49
  3979.4 1808.66  4043.2 1808.62    4154 1806.42  4194.3 1806.83  4234.5 1804.47
  4274.7  1805.1  4311.2 1803.77  4316.2 1804.34    4345 1803.62  4385.1 1805.49
  4836.9 1805.49  4917.2 1804.22  4957.4 1801.24    4990 1801.08  5000.7 1799.85
  5001.2 1799.35  5014.5 1799.85  5037.7 1804.06    5118 1804.56  5207.9 1807.64
  5238.5 1807.56  5248.5 1808.63  5268.6 1808.66  5419.2 1814.59  5544.7 1815.15
#Mann= 3 ,-1 , 0
  3471.5     .05       0  5000.7     .05       0  5014.5     .05       0
Bank Sta=5000.7,5014.5
XS Rating Curve= 0 ,0
Exp/Cntr=0.3,0.1

Type RM Length L Ch R = 1 ,30626   ,572,572,572
BEGIN DESCRIPTION:
Mapping XS 67707f6f
END DESCRIPTION:
XS GIS Cut Line= 3
      1577844.45      6817735.42        1579025.      6817822.22
       1580038.9      6817961.11
#Sta/Elev= 30
  3510.3  1815.9  3791.6 1811.02  4232.8    1806  4291.7 1804.94  4296.8 1803.45
    4313 1803.86  4383.2 1802.79  4413.3 1803.72  4453.4 1803.13  4771.6 1803.54
  4855.5 1801.29  4986.7  1801.9  4993.1 1801.67  4998.2 1800.12  5010.1 1799.46
  5010.6 1798.96  5023.4 1798.96  5023.9 1799.46  5057.4 1800.13  5065.3 1800.86
  5070.4 1803.09  5097.8 1804.47  5249.2 1807.32  5269.4 1806.75  5286.9  1807.7
  5400.6  1807.1  5531.8 1808.84  5585.6 1808.46    5663 1810.24  5717.4 1810.05
#Mann= 3 ,-1 , 0
  3510.3     .05       0  5010.1     .05       0  5023.9     .05       0
Bank Sta=5010.1,5023.9
XS Rating Curve= 0 ,0
Exp/Cntr=0.3,0.1

Type RM Length L Ch R = 1 ,30054   ,471,471,471
BEGIN DESCRIPTION:
Mapping XS 60ba8b53
END DESCRIPTION:
XS GIS Cut Line= 3
      1577636.12      6818155.56      1578781.95      6818235.42
      1579858.34      6818398.61
#Sta/Elev= 30
  3563.8 1814.97  3592.7 1815.11  3816.5 1810.16    4094 1807.91    4114 1808.49
  4144.1 1807.54  4174.2 1808.13  4274.4 1806.64  4575.1 1798.65  4655.3  1801.3
    4674 1800.99    4679 1799.79    4762 1801.46  4857.1  1800.8  4988.6 1803.41
  4998.7 1801.38  5001.9 1797.53  5002.4 1797.03  5015.7 1797.53  5018.9 1800.07
  5026.9 1802.28  5039.1 1803.35  5049.3 1802.65  5159.4 1802.97  5403.3 1804.97
  5453.8 1804.99  5474.1 1803.89  5544.9 1806.35  5635.9 1805.61  5801.1 1806.79
#Mann= 3 ,-1 , 0
  3563.8     .05       0  5001.9     .05       0  5015.7     .05       0
Bank Sta=5001.9,5015.7
XS Rating Curve= 0 ,0
Exp/Cntr=0.3,0.1

Type RM Length L Ch R = 1 ,29583   ,447,447,447
BEGIN DESCRIPTION:
Mapping XS 56fe1b57
END DESCRIPTION:
XS GIS Cut Line= 3
      1577726.42      6818596.53      1578636.11      6818665.97
      1579667.32      6818815.27
#Sta/Elev= 30
  3788.4 1814.98    3807 1815.03  3827.1 1812.98  3897.3 1810.06  3957.5 1809.43
  4003.7  1807.3  4358.6 1800.93  4438.9 1801.11  4527.2 1798.55  4663.1 1799.07
  4672.7 1796.58  4673.2 1796.08  4686.5 1796.58  4697.7 1799.06  4709.7 1799.52
  4861.3 1798.35  4982.5 1801.09  5002.7 1798.07    5023 1799.08  5028.5 1801.11
  5033.5 1801.19  5275.6 1800.83  5304.5 1802.62  5356.4 1802.03  5538.3 1804.24
  5578.7 1803.66  5649.4 1804.45  5655.8 1805.76  5669.6 1806.05  5742.7 1805.21
#Mann= 3 ,-1 , 0
  3788.4     .05       0  4672.7     .05       0  4686.5     .05       0
Bank Sta=4672.7,4686.5
XS Rating Curve= 0 ,0
Exp/Cntr=0.3,0.1

Type RM Length L Ch R = 1 ,29136   ,312,312,312
BEGIN DESCRIPTION:
Mapping XS 0c3fb161
END DESCRIPTION:
XS GIS Cut Line= 3
      1577736.33       6818999.3      1578237.67      6819092.62
      1579528.88      6819146.87
#Sta/Elev= 30
  3922.3 1816.16  3961.6 1815.01  4002.3 1812.48  4022.7 1812.58    4043 1810.18
  4134.6 1807.07  4175.2 1806.88  4213.3 1805.19  4323.9 1803.12  4419.4 1802.49
  4469.6 1800.75  4689.8 1798.08  4729.8 1797.04  4732.9  1796.2  4733.4  1795.7
  4746.7  1796.2  4759.9 1797.99  4779.9  1796.6  4799.9 1797.77  4883.6 1798.01
  4982.6 1799.47  4990.1 1798.84  5000.1 1796.34  5040.1 1799.16  5180.2 1798.82
  5240.3 1800.29  5510.5 1801.29    5634 1803.07  5660.7  1804.5  5724.6 1804.67
#Mann= 5 ,-1 , 0
  3922.3     .05       0  4732.9     .05       0  4746.7     .05       0
  4883.6     .12       0  4982.6     .05       0
Bank Sta=4732.9,4746.7
XS Rating Curve= 0 ,0
Exp/Cntr=0.3,0.1

Type RM Length L Ch R = 1 ,28824   ,420,420,420
BEGIN DESCRIPTION:
Mapping XS 1759900f
END DESCRIPTION:
XS GIS Cut Line= 3
      1577671.26      6819251.04      1578300.61      6819379.08
      1579600.26      6819376.91
#Sta/Elev= 30
  3813.9 1815.17  3838.1 1814.28  3848.3 1814.85  3873.9 1813.08    3930 1812.03
  3950.4 1810.32  4001.4 1809.46  4042.2 1807.28  4134.1 1804.96  4455.8 1799.06
  4550.5 1798.73  4580.5 1797.79  4600.5 1798.38  4870.5 1797.07  4940.5 1798.17
  4963.1 1796.98  4963.6 1796.48  4977.9 1796.98  5090.5 1798.64  5140.5 1798.06
  5150.5 1799.15  5190.5 1799.48  5330.5 1799.48  5360.5 1800.21  5390.5 1802.81
  5440.5 1800.31  5600.5 1802.79  5660.5 1802.75  5740.5 1804.29  5755.8 1806.51
#Mann= 3 ,-1 , 0
  3813.9     .05       0  4963.1     .05       0  4977.9     .05       0
Bank Sta=4963.1,4977.9
XS Rating Curve= 0 ,0
Exp/Cntr=0.3,0.1

Type RM Length L Ch R = 1 ,28404   ,760,760,760
BEGIN DESCRIPTION:
Mapping XS aab38d50
END DESCRIPTION:
XS GIS Cut Line= 3
       1577653.9      6819576.56      1578476.39      6819767.54
      1579500.39      6819808.76
#Sta/Elev= 30
  3826.8 1809.65  3848.5 1809.08  3859.6 1810.11  3902.2 1807.45  3961.4 1807.16
  3987.5 1805.42    4064 1804.55  4120.5 1802.63  4381.5 1799.12  4464.4 1799.19
    4485 1797.96    4526 1798.49  4556.8 1797.47  4567.5  1794.9  4569.9  1793.3
  4570.4  1792.8  4584.7  1793.3  4618.4 1796.08  4652.7 1795.43  4749.8 1796.69
  4769.9 1797.79  4789.9  1795.8  4799.9 1795.78    4811 1797.81    4920 1795.43
    4960 1796.51    5000 1795.43  5460.4 1798.79  5680.6 1803.68    5696 1804.74
#Mann= 3 ,-1 , 0
  3826.8     .05       0  4569.9     .05       0  4584.7     .05       0
Bank Sta=4569.9,4584.7
XS Rating Curve= 0 ,0
Exp/Cntr=0.3,0.1

Type RM Length L Ch R = 1 ,27644   ,508,508,508
BEGIN DESCRIPTION:
Mapping XS df1be954
END DESCRIPTION:
XS GIS Cut Line= 4
      1577623.49      6819912.92      1578476.39      6820216.75
      1579285.85      6820284.03      1579550.34      6820247.17
#Sta/Elev= 30
  3700.6 1804.09  4027.3 1798.61  4114.5 1798.74  4181.4 1797.46  4263.3 1797.81
  4424.1 1795.47  4535.4 1795.83  4560.9    1797  4583.3 1794.24  4602.6 1796.59
  4624.7 1795.82  4634.7 1796.56  4815.3 1796.51  4955.8  1795.4    4996 1792.41
  4998.5 1791.48    4999 1790.98  5013.4 1791.48    5016 1792.78  5036.1 1794.48
  5096.3 1795.67  5116.4 1794.56  5206.7 1795.22    5283 1797.25  5347.2 1796.81
  5467.9 1798.93  5629.4 1803.74  5659.7 1806.46  5682.6 1806.83  5685.3 1806.85
#Mann= 5 ,-1 , 0
  3700.6     .05       0  4998.5     .05       0  5013.4     .05       0
    5283    .075       0  5682.6     .05       0
Bank Sta=4998.5,5013.4
XS Rating Curve= 0 ,0
Exp/Cntr=0.3,0.1

Type RM Length L Ch R = 1 ,27136   ,1087,1087,1087
BEGIN DESCRIPTION:
Mapping XS 67269d83
END DESCRIPTION:
XS GIS Cut Line= 4
      1577569.27      6820320.92      1578597.92      6820520.57
      1579190.37      6820728.91      1579421.26       6820754.8
#Sta/Elev= 30
  3658.7 1800.64  3756.2 1798.96  3970.1 1797.94  4036.7 1798.14  4041.8 1799.48
    4072  1797.9  4088.4 1799.47  4093.5 1798.18  4112.7 1797.53  4418.3 1793.22
  4455.4 1793.92  4489.7 1792.56  4499.8 1793.48  4563.9 1792.54  4711.3 1794.48
  4897.1 1794.12  4953.8  1795.2  4979.1 1792.35  4992.8 1789.48  4993.3 1788.98
  5007.7 1789.48  5010.4 1789.65  5015.7 1792.91  5021.5 1794.67  5032.1 1796.37
  5116.9 1793.91  5307.7 1795.33  5429.8 1800.26    5458 1799.33  5566.9 1801.18
#Mann= 3 ,-1 , 0
  3658.7     .05       0  4992.8     .05       0  5007.7     .05       0
Bank Sta=4992.8,5007.7
XS Rating Curve= 0 ,0
Exp/Cntr=0.3,0.1

Type RM Length L Ch R = 1 ,26049   ,160,160,160
BEGIN DESCRIPTION:
Mapping XS 126a32fc
END DESCRIPTION:
XS GIS Cut Line= 4
      1577122.23      6820943.75      1578022.83      6820971.96
      1578801.91      6820917.71      1579288.06      6820798.34
#Sta/Elev= 30
  3915.2 1801.15  3939.8  1799.8  3945.5 1799.59    4018 1798.41    4058 1798.82
  4206.9  1797.1  4228.1 1797.92  4288.2  1796.2  4341.3 1796.39  4398.2 1797.01
  4440.2 1796.44  4608.3 1794.67  4638.3 1794.93  4737.1 1792.93  4848.5 1792.58
  4949.5 1789.62  4978.8 1791.34  5001.2 1789.14  5001.7 1788.64  5016.1 1788.64
  5016.6 1789.14  5028.9 1790.76  5086.6  1792.1  5632.6 1793.54  5706.7 1794.06
  5782.6 1794.06  5995.6 1795.91  6037.2 1796.78  6053.5 1799.17  6097.8 1800.68
#Mann= 10 ,-1 , 0
  3915.2     .05       0  3939.8    .075       0  3945.5     .05       0
  4341.3    .075       0  4440.2     .05       0  4737.1    .075       0
  5001.2     .07       0  5016.6    .075       0  5632.6    .075       0
  5706.7     .05       0
Bank Sta=5001.2,5016.6
XS Rating Curve= 0 ,0
Exp/Cntr=0.3,0.1

Type RM Length L Ch R = 1 ,25889   ,483,483,483
BEGIN DESCRIPTION:
Mapping XS 02714200
END DESCRIPTION:
XS GIS Cut Line= 3
      1577443.85      6821115.63      1577909.12      6821126.04
      1578777.14      6821103.47
#Sta/Elev= 30
  4240.1 1798.08  4271.3 1796.08  4291.3 1796.44  4301.3 1795.55  4462.9  1794.4
  4480.6 1794.32  4761.4 1792.45  4871.4 1790.96  4921.4 1791.36  4951.5 1790.42
  4983.8 1787.84  4984.3 1787.34  4999.2 1787.84  5012.9 1789.59  5061.5 1791.77
    5093 1794.08  5131.5 1794.97  5191.5 1794.95  5201.5  1793.6  5206.9 1791.71
  5211.9 1792.08  5221.5 1791.21  5251.6 1791.97  5271.6 1794.11  5330.3 1794.66
  5451.6  1794.1  5466.1 1794.81  5491.6 1796.36  5511.6 1794.22  5573.8 1796.52
#Mann= 9 ,-1 , 0
  4240.1    .075       0  4462.9     .05       0  4480.6    .075       0
  4983.8     .07       0  4999.2    .075       0  5012.9     .05       0
    5093    .075       0  5330.3     .05       0  5466.1    .075       0
Bank Sta=4983.8,4999.2
XS Rating Curve= 0 ,0
Exp/Cntr=0.3,0.1

Type RM Length L Ch R = 1 ,25406   ,275,275,275
BEGIN DESCRIPTION:
Mapping XS 9283d0a7
END DESCRIPTION:
XS GIS Cut Line= 5
      1577711.32      6821378.22      1578062.87      6821534.46
      1578169.21      6821527.95      1578173.55      6821527.95
      1578186.56      6821523.61
#Sta/Elev= 30
  4769.8 1798.54  4803.7 1798.27  4817.6  1798.8  4826.9  1798.3  4832.4 1796.64
  4850.2 1795.73  4855.7 1793.72  4861.4 1793.19  4884.4 1791.82  4916.1 1790.97
  4948.7 1788.74  4982.9 1788.27  5000.7 1788.59  5006.1 1788.23  5021.6 1784.87
  5022.1 1784.37  5036.6 1784.37  5037.1 1784.87  5047.2 1789.38  5058.4 1791.21
  5069.3 1791.75  5081.4 1791.58  5099.2 1790.41  5104.6  1790.7  5122.4 1790.01
  5206.7 1790.09  5226.8 1790.81  5236.8  1792.1  5256.4 1795.59  5279.1 1795.73
#Mann= 3 ,-1 , 0
  4769.8     .05       0  5021.6     .03       0  5037.1     .05       0
Bank Sta=5021.6,5037.1
XS Rating Curve= 0 ,0
Exp/Cntr=0.3,0.1

Type RM Length L Ch R = 1 ,25131   ,200,200,200
BEGIN DESCRIPTION:
Mapping XS 2c882516
END DESCRIPTION:
XS GIS Cut Line= 3
      1577515.97      6821712.41      1577715.65      6821740.63
      1578238.61      6821666.85
#Sta/Elev= 30
  4656.4 1793.81  4665.6 1794.25  4726.1 1793.62  4766.5 1792.25  4807.8 1791.76
  4827.1 1792.01  4847.3 1792.97  4860.3 1792.85  4877.6 1790.54  4928.1 1788.48
  4938.2 1787.19  4948.3 1784.82  5047.2 1784.81  5047.7 1784.31  5062.5 1784.31
    5063 1784.81  5069.5 1784.81  5079.6 1788.39  5089.7 1789.77  5099.8 1790.39
  5131.3 1790.94  5160.4 1790.51  5197.4 1789.15  5241.2 1789.61  5261.4 1788.85
  5281.6 1789.58  5344.7 1788.98  5362.4 1790.23  5372.5 1793.81  5386.2 1794.43
#Mann= 3 ,-1 , 0
  4656.4     .05       0  5047.2     .03       0    5063     .05       0
Bank Sta=5047.2,5063
XS Rating Curve= 0 ,0
Exp/Cntr=0.3,0.1

Type RM Length L Ch R = 1 ,24931   ,270,270,270
BEGIN DESCRIPTION:
Mapping XS 74fd1e86
END DESCRIPTION:
XS GIS Cut Line= 2
      1577750.39      6822005.37      1578275.51      6821705.92
#Sta/Elev= 30
    4770 1794.21  4786.8 1793.95  4799.5 1792.33  4815.4 1790.93  4852.8 1790.58
  4858.6 1790.09  4874.4 1789.86  4880.2 1789.22  4890.3 1789.21  4901.9 1787.69
  4903.9 1784.75  4904.4 1784.25  4919.3 1784.25  4919.8 1784.75  5094.8 1784.76
  5100.6 1785.13  5109.1 1787.91  5116.4 1788.22  5132.2 1788.56  5166.7 1787.69
  5197.1 1789.06  5224.5 1789.78  5283.5 1789.25  5293.3 1788.47  5315.2 1788.43
  5327.9 1789.08  5336.8 1790.06  5350.9 1794.13  5364.2 1794.98  5374.5    1795
#Mann= 3 ,-1 , 0
    4770     .05       0  4903.9     .03       0  4919.8     .05       0
Bank Sta=4903.9,4919.8
XS Rating Curve= 0 ,0
Exp/Cntr=0.3,0.1

Type RM Length L Ch R = 1 ,24661   ,297,297,297
BEGIN DESCRIPTION:
Mapping XS d721c8f4
END DESCRIPTION:
XS GIS Cut Line= 3
      1577798.15        6822307.      1578190.91      6822009.72
      1578290.38      6821765.37
#Sta/Elev= 30
  4729.7 1791.46  4798.7  1791.5  4804.9 1790.89  4834.1 1789.64  4854.9 1789.76
  4869.4 1789.09    4876 1784.67  4876.5 1784.17  4891.4 1784.17  4891.9 1784.67
  5112.9 1784.69  5127.1  1788.2  5133.7 1788.43    5219 1788.41  5267.3 1788.75
  5288.9 1789.37  5302.3 1788.86  5320.9 1788.95  5332.1 1788.08  5342.9 1787.95
  5364.5 1789.06  5374.5 1788.92  5379.9 1787.76  5403.9 1788.02  5418.5 1788.79
  5457.4 1789.26  5462.8 1790.13  5472.5 1793.01  5481.5 1795.03  5486.1 1795.07
#Mann= 3 ,-1 , 0
  4729.7     .05       0    4876     .03       0  4891.9     .05       0
Bank Sta=4876,4891.9
XS Rating Curve= 0 ,0
Exp/Cntr=0.3,0.1

Type RM Length L Ch R = 1 ,24364   ,87,87,87
BEGIN DESCRIPTION:
Mapping XS 8044fc9d
END DESCRIPTION:
XS GIS Cut Line= 4
      1578201.76      6822641.21      1578236.48      6822374.31
      1578219.12      6822037.93      1578312.44      6821784.01
#Sta/Elev= 30
  4618.5 1789.67  4623.3 1789.68  4684.8 1790.18  4702.4 1788.52  4732.7 1786.78
  4763.9 1789.25  4783.1 1788.88  4793.2 1789.91    4838 1788.56  4853.7  1787.5
  4887.6 1788.64    4904 1790.24    4914 1788.91  4916.1 1784.65  4916.6 1784.15
  4931.5 1784.15    4932 1784.65  5094.2 1784.65  5104.2 1785.28  5114.3 1788.72
  5134.3 1788.52  5194.4 1789.84  5330.9 1788.62  5344.9 1787.55  5400.6 1788.13
  5405.9 1788.77  5456.2 1789.73  5461.5 1792.52  5469.4 1794.48    5495 1794.69
#Mann= 4 ,-1 , 0
  4618.5    .075       0  4623.3     .05       0  4916.1     .03       0
    4932     .05       0
Bank Sta=4916.1,4932
XS Rating Curve= 0 ,0
Exp/Cntr=0.3,0.1

Type RM Length L Ch R = 1 ,24277   ,283,283,283
BEGIN DESCRIPTION:
Mapping XS 3340c2d6
END DESCRIPTION:
XS GIS Cut Line= 3
      1578340.65      6822632.55       1578292.9      6822020.57
      1578334.14      6821807.87
#Sta/Elev= 30
  4604.4 1788.59  4659.1 1788.74  4699.2 1787.76  4719.3 1786.39  4737.8  1787.2
  4749.4 1789.38  4759.4 1789.79  4809.6 1786.82  4839.7 1785.92  4859.7 1786.51
  4899.8 1789.49  4909.9 1788.18  4919.9 1780.11    4922 1780.08  4922.5 1779.58
  4937.4 1779.58  4937.9 1780.08  5040.3 1780.08  5050.3 1784.99  5060.3 1787.62
  5070.4 1787.92  5170.7 1789.66  5271.8  1788.1  5292.2 1787.21  5307.7 1788.73
  5312.8 1788.25  5364.6 1788.96  5373.7 1789.69    5394 1792.98  5434.9 1794.43
#Mann= 3 ,-1 , 0
  4604.4     .05       0    4922     .03       0  4937.9     .05       0
Bank Sta=4922,4937.9
XS Rating Curve= 0 ,0
Exp/Cntr=0.3,0.1

Type RM Length L Ch R = 1 ,23994   ,339,339,339
BEGIN DESCRIPTION:
Mapping XS 6eef8ac6
END DESCRIPTION:
XS GIS Cut Line= 3
      1578381.87      6822660.79        1578664.      6822107.38
      1578755.14      6821877.36
#Sta/Elev= 30
  4557.2 1788.78  4681.7 1788.94  4703.9 1789.64  4717.5 1788.96  4726.2 1786.61
  4776.2 1786.76  4792.9 1787.93  4820.7    1786  4842.9 1785.33  4964.4 1785.87
  4976.3 1784.32  4978.9 1780.07  4979.4 1779.57  4994.3 1779.57  4994.8 1780.07
  5065.4 1780.07  5076.3 1784.75  5098.5 1786.38  5126.4 1786.93    5143 1789.39
  5165.2 1789.73  5175.2 1788.37  5199.6 1788.12  5302.3 1789.81  5307.7 1790.08
  5317.5 1792.56  5326.7  1793.9  5339.1 1794.28  5386.1 1794.57  5425.8 1793.78
#Mann= 3 ,-1 , 0
  4557.2     .05       0  4978.9     .03       0  4994.8     .05       0
Bank Sta=4978.9,4994.8
XS Rating Curve= 0 ,0
Exp/Cntr=0.3,0.1

Type RM Length L Ch R = 1 ,23655   ,421,421,421
BEGIN DESCRIPTION:
Mapping XS 82207c9d
END DESCRIPTION:
XS GIS Cut Line= 3
      1578427.43      6822728.06      1578520.77      6822630.38
      1579138.57      6822402.77
#Sta/Elev= 30
  4669.7 1788.84  4731.4 1788.39  4804.8 1789.64  4841.3 1789.44  4850.9 1786.91
  4862.6 1785.59  4886.6 1786.25  4911.7 1785.24  4917.1 1785.72  4936.9 1783.61
  4942.2 1781.04  4947.9 1780.04  4989.8 1780.04  4990.3 1779.54  5005.3 1779.54
  5005.8 1780.04  5022.5 1780.04  5043.8 1785.35  5065.1 1785.83  5075.7  1785.3
  5097.1 1785.43    5129 1787.23  5175.1 1786.73    5193 1786.02  5246.3 1786.16
  5310.2 1788.99  5408.1  1790.7  5438.5 1792.28  5448.7 1793.55  5463.2 1796.85
#Mann= 4 ,-1 , 0
  4669.7    .075       0  4731.4     .05       0  4989.8     .03       0
  5005.8     .05       0
Bank Sta=4989.8,5005.8
XS Rating Curve= 0 ,0
Exp/Cntr=0.3,0.1

Type RM Length L Ch R = 1 ,23234   ,405,405,405
BEGIN DESCRIPTION:
Mapping XS 2d9c86be
END DESCRIPTION:
XS GIS Cut Line= 3
      1578342.85      6823012.32      1578826.76      6822936.37
      1579194.81      6822782.66
#Sta/Elev= 30
  4337.2 1786.66  4420.4 1785.14  4526.5 1785.12  4582.3 1783.13  4656.8 1783.58
  4693.7 1782.89  4734.2 1783.61  4787.1 1786.76  4833.2 1786.65  4840.7 1787.99
  4862.4 1789.46  4883.8 1786.06  4915.4 1784.24  4944.7 1784.38  4955.2 1783.73
  4976.8 1779.99  4992.3 1779.99  5008.1 1779.99  5008.6 1779.49  5024.1 1779.99
  5042.4 1779.99  5052.7 1781.77  5063.5 1784.88  5069.1 1787.31    5093 1787.91
  5098.4 1789.05    5146 1789.16  5175.2 1787.07  5182.8 1788.36  5225.9 1789.51
#Mann= 7 ,-1 , 0
  4337.2     .05       0  4840.7     .12       0  4883.8     .05       0
  4992.3     .12       0  5008.1     .07       0  5024.1     .12       0
  5042.4     .05       0
Bank Sta=5008.1,5024.1
XS Rating Curve= 0 ,0
Exp/Cntr=0.3,0.1

Type RM Length L Ch R = 1 ,22829   ,307,307,307
BEGIN DESCRIPTION:
Mapping XS 2a6bbc22
END DESCRIPTION:
XS GIS Cut Line= 2
       1578614.1      6823257.55      1579441.54      6823227.23
#Sta/Elev= 30
  4608.6 1786.54  4649.5 1785.99  4659.5 1785.48  4689.6 1782.77  4709.6 1782.26
  4739.6  1782.6  4779.6 1783.78  4839.7 1783.59  4859.7 1783.34  4869.7 1780.38
  4879.7 1779.97  5051.5 1779.96    5052 1779.46  5067.7 1779.46  5068.2 1779.96
  5069.8 1781.28  5079.8 1784.55  5089.8 1785.76  5099.8 1786.19  5159.9 1784.98
  5169.9 1785.12  5249.9 1789.17  5269.9 1788.81    5277 1788.06    5320  1787.9
    5360 1789.03    5370 1790.71    5380 1791.42    5420 1791.36  5436.6 1790.93
#Mann= 3 ,-1 , 0
  4608.6     .05       0  5051.5     .05       0  5068.2     .05       0
Bank Sta=5051.5,5068.2
XS Rating Curve= 0 ,0
Exp/Cntr=0.3,0.1
