HEC-RAS study Buttonwillow Creek.prj: Buttonwillow Creek Base Level Engineering

--- Buttonwillow Creek.g01 (geometry) --- (continued)

Type RM Length L Ch R = 1 ,22522   ,252,252,252
BEGIN DESCRIPTION:
Mapping XS 98c63d16
END DESCRIPTION:
XS GIS Cut Line= 3
      1578633.64      6823591.75      1578854.97      6823574.39
      1579555.89      6823459.38
#Sta/Elev= 30
  4615.1  1785.8  4636.5 1786.41  4676.6 1784.56  4686.7  1784.6  4696.7 1785.04
  4746.9 1785.28    4777 1785.26    4807 1784.81  4839.7 1783.74    4849  1783.1
  4857.4 1779.91    5072  1779.9  5072.5  1779.4  5088.2  1779.4  5088.7  1779.9
    5131  1779.9  5141.1 1782.46  5161.4 1783.28  5211.6 1783.56    5278 1785.27
  5313.4 1785.89  5339.3  1785.6  5344.3  1785.9  5394.5 1786.54  5414.8 1787.55
    5435 1789.23  5445.2 1789.71  5466.9 1789.71  5485.7 1790.05  5547.4  1789.4
#Mann= 3 ,-1 , 0
  4615.1     .05       0    5072     .03       0  5088.7     .05       0
Bank Sta=5072,5088.7
XS Rating Curve= 0 ,0
Exp/Cntr=0.3,0.1

Type RM Length L Ch R = 1 ,22270   ,54,54,54
BEGIN DESCRIPTION:
Mapping XS ea1e307c
END DESCRIPTION:
XS GIS Cut Line= 3
      1578695.24      6823753.43      1579053.27      6823759.94
      1579630.84      6823707.93
#Sta/Elev= 30
  4541.1 1784.86  4590.9 1785.04  4600.9  1784.5  4610.9 1782.62  4640.9 1782.13
  4700.9 1782.29  4840.9 1784.34  4880.9 1783.33    4921 1784.51  4941.1 1779.86
  4962.9 1779.86  4963.4 1779.36  4979.1 1779.36  4979.6 1779.86  5021.4 1779.86
  5031.5 1782.89  5041.5 1784.19  5121.8 1785.08    5162    1785  5212.2 1786.13
  5242.3 1785.81  5302.6 1786.72  5332.7 1786.51  5342.7 1786.72  5352.8 1787.96
  5362.8 1788.27  5425.3 1789.13  5453.2 1788.93  5473.2 1788.43  5479.1  1787.8
#Mann= 3 ,-1 , 0
  4541.1     .05       0  4962.9     .03       0  4979.6     .05       0
Bank Sta=4962.9,4979.6
XS Rating Curve= 0 ,0
Exp/Cntr=0.3,0.1

Type RM Length L Ch R = 1 ,22216   ,275,275,275
BEGIN DESCRIPTION:
Mapping XS fb6b2c9f
END DESCRIPTION:
XS GIS Cut Line= 3
      1578687.57      6823823.96      1579068.46      6823809.85
      1579624.01      6823771.88
#Sta/Elev= 30
  4532.6 1785.31  4590.1 1785.12  4600.1 1784.03  4610.1 1781.78  4710.2 1781.39
    4832 1783.57  4900.3 1782.94  4920.3 1784.79  4930.3 1783.35  4940.4 1778.77
    4942 1776.58  4942.5 1776.08  4958.2 1776.08  4958.7 1776.58  5014.9 1776.58
  5020.5  1778.7  5030.6 1780.12  5040.6 1783.71  5050.6 1784.75  5060.6 1785.01
  5100.7  1784.2  5158.4 1784.43  5180.9 1785.05    5211 1786.93    5231 1785.33
  5261.1 1784.97  5371.4 1786.87  5391.4 1788.22  5411.5 1788.69  5470.6 1788.47
#Mann= 3 ,-1 , 0
  4532.6     .05       0    4942     .03       0  4958.7     .05       0
Bank Sta=4942,4958.7
XS Rating Curve= 0 ,0
Exp/Cntr=0.3,0.1

Type RM Length L Ch R = 1 ,21941   ,369,369,369
BEGIN DESCRIPTION:
Mapping XS 66fb4c77
END DESCRIPTION:
XS GIS Cut Line= 2
      1578700.59      6824083.29      1579848.64      6824072.44
#Sta/Elev= 30
    4546 1785.18  4570.4 1784.94  4581.1  1785.3  4590.4 1784.86  4620.4 1781.89
  4660.4 1781.08  4710.4 1781.21  4790.4 1780.35  4820.4 1778.36  4821.9 1776.58
  4822.4 1776.08  4838.4 1776.08  4838.9 1776.58  5210.4 1776.58  5220.4 1781.19
  5240.4 1783.51  5290.4 1786.16  5310.4 1785.69  5330.4 1785.95  5350.4 1788.21
  5370.4 1788.95  5440.4 1788.79  5490.4 1787.62  5500.4 1787.99  5520.4 1787.64
  5540.5 1789.14  5550.5 1790.49  5580.5 1792.18  5630.1  1792.2  5694.1 1793.15
#Mann= 3 ,-1 , 0
    4546     .05       0  4821.9     .03       0  4838.9     .05       0
Bank Sta=4821.9,4838.9
XS Rating Curve= 0 ,0
Exp/Cntr=0.3,0.1

Type RM Length L Ch R = 1 ,21572   ,271,271,271
BEGIN DESCRIPTION:
Mapping XS 99d52b1d
END DESCRIPTION:
XS GIS Cut Line= 2
      1578720.76      6824466.45       1579774.6      6824421.31
#Sta/Elev= 30
  4565.7 1784.31    4610 1783.92    4620 1781.81    4640 1780.65  4700.1 1781.55
  4730.1 1779.95  4770.1 1781.25  4810.2  1783.9  4890.2 1784.09  4910.3 1782.78
  4920.3 1780.98  4921.7 1776.58  4922.2 1776.08  4938.8 1776.58  5070.4 1776.58
  5080.4 1778.29  5090.4 1782.21  5109.5 1785.73  5114.6 1784.62  5130.5 1786.36
  5160.5 1786.59  5260.6 1790.51  5330.6 1790.02  5346.5 1788.93  5390.7 1788.68
  5400.7 1788.83  5430.7 1791.57  5470.8 1793.03  5510.8 1792.73  5620.5 1794.34
#Mann= 3 ,-1 , 0
  4565.7     .05       0  4921.7     .03       0  4938.8     .05       0
Bank Sta=4921.7,4938.8
XS Rating Curve= 0 ,0
Exp/Cntr=0.3,0.1

Type RM Length L Ch R = 1 ,21301   ,158,158,158
BEGIN DESCRIPTION:
Mapping XS 06257182
END DESCRIPTION:
XS GIS Cut Line= 3
      1578718.99      6824707.77      1579062.77      6824714.71
      1579671.07      6824700.85
#Sta/Elev= 30
  4539.3 1783.25  4565.3 1783.69  4665.3 1783.12  4705.3  1783.8  4735.3 1783.54
  4765.4 1783.85  4794.3 1783.51  4805.4 1782.58  4815.4 1782.42  4825.4 1783.13
  4855.4 1783.88  4895.4 1783.31  4915.4 1783.54  4935.4 1781.48  4945.4 1777.73
  4945.8 1776.58  4946.3 1776.08  4962.4 1776.08  4962.9 1776.58  5065.4 1776.58
  5085.4  1782.7  5095.4 1783.83  5165.4 1784.54  5195.5 1784.19  5235.5 1786.63
  5315.5 1789.46  5335.5 1787.96  5365.5 1788.48  5405.5 1792.06  5491.6 1792.35
#Mann= 3 ,-1 , 0
  4539.3     .05       0  4945.8     .05       0  4962.9     .05       0
Bank Sta=4945.8,4962.9
XS Rating Curve= 0 ,0
Exp/Cntr=0.3,0.1

Type RM Length L Ch R = 1 ,21143   ,170,170,170
BEGIN DESCRIPTION:
Mapping XS 91d7a404
END DESCRIPTION:
XS GIS Cut Line= 3
      1578574.95      6824883.12      1579074.93      6824867.49
      1579757.25      6824839.71
#Sta/Elev= 30
  4369.7  1782.4  4449.8 1783.04  4629.9 1782.14  4689.2 1782.72  4729.9 1781.47
    4810 1782.16    4920 1781.91    4930 1781.58    4940  1779.5  4961.3 1772.57
  4961.8 1772.07  4978.4 1772.07  4978.9 1772.57  5020.1    1773  5040.1 1780.68
  5050.1 1782.05  5060.1  1782.1  5080.2 1781.32  5110.2 1782.82  5170.2 1783.26
  5210.3 1784.48  5225.7    1784  5240.3 1784.28  5290.3 1786.38  5320.4 1786.84
  5330.4 1788.57  5360.4 1789.41  5430.5 1789.87  5468.7 1790.83  5552.8 1790.88
#Mann= 3 ,-1 , 0
  4369.7     .05       0  4961.3     .05       0  4978.9     .05       0
Bank Sta=4961.3,4978.9
XS Rating Curve= 0 ,0
Exp/Cntr=0.3,0.1

Type RM Length L Ch R = 1 ,20973   ,428,428,428
BEGIN DESCRIPTION:
Mapping XS 99af9588
END DESCRIPTION:
XS GIS Cut Line= 2
      1578647.82      6825048.05       1579660.9      6825018.56
#Sta/Elev= 30
  4442.5 1780.86  4459.7  1781.2  4489.7 1780.37  4629.8 1780.18  4639.8 1780.21
  4649.8  1780.9  4669.8  1780.2  4779.8 1781.29  4819.8 1780.82  4849.8 1781.14
  4919.9 1779.27  4929.9 1779.73  4949.9 1779.03  4957.3  1777.7  4962.3 1777.52
  4979.9 1773.91  4991.1 1772.61  4991.6 1772.11  5008.2 1772.11  5008.7 1772.61
  5039.9 1778.38  5059.9 1778.83    5160 1784.56    5210 1785.16    5260 1784.68
    5280 1785.29  5299.2 1786.62  5304.2 1786.17  5370.1 1788.17    5456 1789.46
#Mann= 3 ,-1 , 0
  4442.5     .05       0  4991.1     .03       0  5008.7     .05       0
Bank Sta=4991.1,5008.7
XS Rating Curve= 0 ,0
Exp/Cntr=0.3,0.1

Type RM Length L Ch R = 1 ,20545   ,475,475,475
BEGIN DESCRIPTION:
Mapping XS dca4b294
END DESCRIPTION:
XS GIS Cut Line= 4
      1578671.24      6825384.62       1578818.8      6825387.12
      1579311.04      6825459.51      1579538.42      6825423.05
#Sta/Elev= 30
  4553.4 1779.31  4647.2 1779.13  4677.2 1779.68    4737 1779.22    4778  1776.3
  4806.7 1775.76  4811.8 1775.93  4818.4 1777.15  4838.6 1779.04  4899.3 1779.35
  4951.2  1777.9  4980.1 1777.79  4990.3 1776.58  5010.5 1772.85  5012.2 1771.78
  5012.7 1771.28  5029.3 1771.28  5029.8 1771.78  5040.8 1772.48  5080.6 1777.91
  5091.3 1777.91  5150.4 1780.94  5212.7 1781.43  5232.9 1780.75  5238.8    1780
  5263.3 1780.81  5283.5  1780.4  5324.1 1781.78  5384.8 1782.98  5428.8 1783.35
#Mann= 3 ,-1 , 0
  4553.4     .05       0  5012.2     .03       0  5029.8     .05       0
Bank Sta=5012.2,5029.8
XS Rating Curve= 0 ,0
Exp/Cntr=0.3,0.1

Type RM Length L Ch R = 1 ,20070   ,335,335,335
BEGIN DESCRIPTION:
Mapping XS 5bcbcc3d
END DESCRIPTION:
XS GIS Cut Line= 3
      1578661.72      6825877.91      1578850.97      6825858.81
      1579154.74       6825872.7
#Sta/Elev= 30
  4683.2 1778.87  4716.7 1779.04  4746.8 1778.19  4756.9 1777.64    4777 1777.75
  4797.1 1777.27    4832 1778.47  4857.4 1778.55  4867.4 1778.88  4907.5 1778.22
  4917.5  1778.3  4937.5 1777.04  4968.8 1776.35  4987.6 1772.42  4997.6  1770.9
  5008.8 1770.28  5009.3 1769.78  5025.9 1769.78  5026.4 1770.28  5027.6 1770.63
  5037.6 1771.82  5057.6 1775.72  5067.6  1777.1  5077.7 1776.83  5087.7 1777.18
  5107.7 1779.56  5117.7 1779.64  5127.7    1779  5137.7 1778.93  5177.5 1779.17
#Mann= 3 ,-1 , 0
  4683.2     .05       0  5008.8     .03       0  5026.4     .05       0
Bank Sta=5008.8,5026.4
XS Rating Curve= 0 ,0
Exp/Cntr=0.3,0.1

Type RM Length L Ch R = 1 ,19735   ,271,271,271
BEGIN DESCRIPTION:
Mapping XS a510139f
END DESCRIPTION:
XS GIS Cut Line= 3
      1578349.28      6826235.54      1579111.38      6826181.73
      1579261.18      6826111.13
#Sta/Elev= 30
  4393.4 1780.27  4426.9 1779.76  4489.4 1779.83    4568 1778.91    4573 1779.18
  4589.6 1778.75  4699.9 1778.26    4730 1778.79    4740 1778.22  4820.2  1777.5
  4900.4 1777.76  4920.4 1777.34  4940.5 1774.93  4980.6 1773.38  4990.6 1772.05
  4996.5 1769.95  5001.5 1769.55  5001.7 1768.75  5002.2 1768.25  5019.1 1768.25
  5019.6 1768.75  5030.7 1769.29  5050.8  1773.6  5080.8 1775.32  5090.9 1777.27
  5100.9 1777.67  5162.2 1778.25  5172.4 1777.65  5251.8 1776.67    5323 1778.77
#Mann= 3 ,-1 , 0
  4393.4    .075       0  5001.7     .07       0  5019.6     .05       0
Bank Sta=5001.7,5019.6
XS Rating Curve= 0 ,0
Exp/Cntr=0.3,0.1

Type RM Length L Ch R = 1 ,19464   ,282,282,282
BEGIN DESCRIPTION:
Mapping XS 2c56d77f
END DESCRIPTION:
XS GIS Cut Line= 3
      1578932.59      6826780.81      1579158.29      6826327.67
      1579301.21      6826136.54
#Sta/Elev= 30
  4541.7 1777.56  4554.4 1777.06  4634.2 1778.06  4666.3 1777.83  4711.1 1776.19
  4723.6 1774.79  4761.4 1775.95  4867.8 1775.29  4873.4 1774.95    4880 1773.45
  4940.5 1772.57  4957.3 1769.53  4960.4 1768.43  4960.9 1767.93  4977.9 1767.93
  4978.4 1768.43  4985.3 1769.74  4991.7 1771.76  5002.1 1773.72    5045 1775.64
  5087.7 1775.82  5096.1 1776.39  5146.1  1776.9  5166.9 1775.84  5181.5  1776.3
  5196.1 1775.87  5216.9  1776.7  5252.4 1776.83  5281.6 1777.69  5286.6 1777.32
#Mann= 3 ,-1 , 0
  4541.7     .05       0  4960.4     .05       0  4978.4     .05       0
Bank Sta=4960.4,4978.4
XS Rating Curve= 0 ,0
Exp/Cntr=0.3,0.1

Type RM Length L Ch R = 1 ,19182   ,299,299,299
BEGIN DESCRIPTION:
Mapping XS 050a5c4a
END DESCRIPTION:
XS GIS Cut Line= 2
      1579357.95      6826871.08      1579382.25      6826263.46
#Sta/Elev= 30
    4617 1776.11    4621 1776.11  4630.1  1776.9  4671.7 1776.59  4690.1 1776.24
  4700.1 1775.67  4770.2 1774.74  4780.2 1773.96  4790.2 1773.66  4820.2 1774.69
  4830.2 1774.41  4850.3 1774.78  4900.3 1774.45  4930.3 1772.17  4950.3 1771.55
  4960.4 1771.97  4970.4 1771.14  4990.4 1767.62  4991.4 1767.01  4991.9 1766.51
  5008.9 1766.51  5009.4 1767.01  5010.4  1767.9  5030.4 1772.56  5050.4  1773.4
  5060.4 1774.93  5110.5 1776.58  5172.1  1776.5  5200.5 1775.79  5225.1 1776.13
#Mann= 3 ,-1 , 0
    4617     .05       0  4991.4     .05       0  5009.4     .05       0
Bank Sta=4991.4,5009.4
XS Rating Curve= 0 ,0
Exp/Cntr=0.3,0.1

Type RM Length L Ch R = 1 ,18883   ,260,260,260
BEGIN DESCRIPTION:
Mapping XS 7372326c
END DESCRIPTION:
XS GIS Cut Line= 4
      1579490.28      6826954.93      1579626.84      6826768.72
      1579666.98      6826577.67      1579698.23      6826037.72
#Sta/Elev= 30
    4484 1775.89  4528.9 1775.53  4564.4 1773.74    4600 1773.29  4606.2 1773.82
  4691.8 1773.69  4736.1 1773.35  4756.5 1772.37  4780.5 1772.91  4797.4 1772.25
  4868.9  1773.7  4912.5 1773.32  4949.9 1771.28  4969.9 1771.17  4979.9    1770
  5000.9 1766.21  5001.4 1765.71  5018.5 1765.71    5019 1766.21    5020 1767.76
    5040 1772.01  5070.1 1773.98  5135.4 1775.78  5169.6 1775.64  5210.3 1774.87
  5230.3 1775.32  5240.4 1774.79  5278.1 1776.17  5410.6 1775.93    5451 1776.75
#Mann= 5 ,-1 , 0
    4484     .05       0  5000.9     .05       0    5019     .05       0
  5169.6    .075       0  5278.1     .05       0
Bank Sta=5000.9,5019
XS Rating Curve= 0 ,0
Exp/Cntr=0.3,0.1

Type RM Length L Ch R = 1 ,18623   ,186,186,186
BEGIN DESCRIPTION:
Mapping XS 9f8ed024
END DESCRIPTION:
XS GIS Cut Line= 4
      1579589.21      6826990.13      1579735.07      6826797.38
       1579913.5      6826596.77       1579986.4      6826162.85
#Sta/Elev= 30
  4379.1 1775.75  4413.3 1773.37  4442.5  1773.3  4448.7 1774.07  4469.6 1772.45
  4513.2 1772.43  4563.2  1771.3  4617.3    1773  4740.4 1772.69  4762.1  1771.5
  4790.5 1772.12  4811.4 1771.37  4854.1 1772.49  4908.3 1772.14    4959 1769.81
  4969.2  1770.1  5000.7 1765.82  5001.2 1765.32  5018.8 1765.82  5019.9 1766.79
  5040.2 1770.37  5052.3 1770.25  5070.6 1772.63  5090.9 1774.08  5212.2 1774.05
  5248.4 1773.83  5283.5 1775.88  5289.6 1775.98  5294.7 1774.85  5329.3 1775.56
#Mann= 5 ,-1 , 0
  4379.1     .05       0  5000.7     .05       0  5018.8     .05       0
  5212.2    .075       0  5248.4     .05       0
Bank Sta=5000.7,5018.8
XS Rating Curve= 0 ,0
Exp/Cntr=0.3,0.1

Type RM Length L Ch R = 1 ,18437   ,210,210,210
BEGIN DESCRIPTION:
Mapping XS 6a4ded46
END DESCRIPTION:
XS GIS Cut Line= 3
        1579683.      6826936.69      1580015.93      6826666.21
      1580361.44      6826200.91
#Sta/Elev= 30
  4450.4 1775.06  4500.9 1774.85  4515.3 1774.01  4521.8 1772.32  4536.1 1771.86
  4550.5 1772.82  4556.9 1771.74  4628.8 1770.78  4635.2 1771.74  4678.4 1772.48
  4785.4  1772.2    4835 1770.96  4855.8 1771.82    4914 1772.12  4976.8 1769.56
  4999.5  1769.5  5014.1 1767.19  5017.5 1765.35    5018 1764.85  5035.7 1765.35
    5064 1769.46  5105.9 1769.96  5141.3 1772.91    5156 1773.39  5291.6 1776.51
  5341.6 1775.55    5350 1774.64  5391.7  1775.1  5420.9 1777.98  5458.9  1778.6
#Mann= 3 ,-1 , 0
  4450.4     .05       0  5017.5     .05       0  5035.7     .05       0
Bank Sta=5017.5,5035.7
XS Rating Curve= 0 ,0
Exp/Cntr=0.3,0.1

Type RM Length L Ch R = 1 ,18227   ,180,180,180
BEGIN DESCRIPTION:
Mapping XS e074b4ad
END DESCRIPTION:
XS GIS Cut Line= 3
       1579694.7      6826940.61      1580132.25      6826740.86
       1580665.2       6826501.3
#Sta/Elev= 30
  4386.1 1775.11  4441.4 1774.63  4455.2 1772.67  4472.8 1774.13  4495.8 1774.35
  4518.3 1774.01  4529.8 1772.79  4547.4  1772.8  4552.9 1772.08  4570.4 1773.02
  4575.9 1771.34  4650.5 1770.69  4719.6 1771.71  4771.2 1770.32  4840.2 1771.42
  4909.6 1770.67  4968.8 1769.26  4992.6 1764.58  4993.1 1764.08  5010.8 1764.58
  5036.3 1768.23  5077.2 1769.39  5105.8 1772.47    5129 1773.46  5188.1 1773.46
  5220.9 1771.89  5250.2 1773.26    5302 1774.13  5325.2 1773.67  5451.4 1774.73
#Mann= 3 ,-1 , 0
  4386.1     .05       0  4992.6     .05       0  5010.8     .05       0
Bank Sta=4992.6,5010.8
XS Rating Curve= 0 ,0
Exp/Cntr=0.3,0.1

Type RM Length L Ch R = 1 ,18047   ,285,285,285
BEGIN DESCRIPTION:
Mapping XS 6b04b833
END DESCRIPTION:
XS GIS Cut Line= 4
      1579809.37      6827020.37      1580196.49      6826893.64
      1580635.73      6826721.77      1580785.04      6826628.01
#Sta/Elev= 30
  4431.2 1775.54  4459.2 1774.29  4485.7 1775.15    4491  1773.8  4517.6 1774.31
  4522.9 1773.25  4581.3 1771.91  4586.6 1773.06  4626.5 1771.39    4714 1771.69
  4763.3 1770.87  4784.4 1769.77  4879.9 1770.98  4949.9  1768.8  4978.2 1763.74
  4978.7 1763.24  4996.4 1763.74  5004.2  1766.2  5019.5 1767.84  5094.7 1770.86
  5105.4 1770.83  5118.1 1769.51  5137.2 1771.29  5212.8 1772.02  5256.5 1771.42
  5275.6 1771.91  5298.7 1771.11    5392  1773.5  5436.4 1773.85  5486.5 1772.21
#Mann= 3 ,-1 , 0
  4431.2     .05       0  4978.2     .05       0  4996.4     .05       0
Bank Sta=4978.2,4996.4
XS Rating Curve= 0 ,0
Exp/Cntr=0.3,0.1

Type RM Length L Ch R = 1 ,17762   ,225,225,225
BEGIN DESCRIPTION:
Mapping XS 36b78d98
END DESCRIPTION:
XS GIS Cut Line= 3
      1580186.05      6827478.74      1580668.71      6826860.66
      1580828.45      6826643.61
#Sta/Elev= 30
    4458 1771.04    4558 1771.12  4593.3 1771.95  4628.6 1771.03  4707.2 1771.24
  4721.7 1770.31  4800.4 1769.77  4870.9 1770.78  4914.4 1769.78  4941.5 1768.16
    4956 1768.45  4970.4 1766.16  4982.7 1763.31  4983.2 1762.81  5000.4 1762.81
  5000.9 1763.31  5005.7 1765.11  5028.3 1767.83  5063.6    1768  5098.9  1771.3
  5119.7  1771.9  5212.8 1770.57  5240.7  1771.9  5262.7 1772.13  5333.7 1772.15
    5363 1771.42  5427.8 1772.49    5434 1771.64  5469.5  1773.2  5511.7 1773.29
#Mann= 3 ,-1 , 0
    4458     .05       0  4982.7     .05       0  5000.9     .05       0
Bank Sta=4982.7,5000.9
XS Rating Curve= 0 ,0
Exp/Cntr=0.3,0.1

Type RM Length L Ch R = 1 ,17537   ,449,449,449
BEGIN DESCRIPTION:
Mapping XS 9d8318c7
END DESCRIPTION:
XS GIS Cut Line= 3
       1580324.9      6827971.89       1580515.5      6827646.53
      1580882.09      6826732.59
#Sta/Elev= 30
    4088 1774.71  4162.6 1772.99  4289.5 1772.14  4324.3 1770.42  4382.2 1770.54
  4440.2 1769.23    4473 1769.85  4610.2 1769.25  4646.7 1770.12  4688.2 1769.71
  4700.5 1768.82  4771.6 1769.21  4786.7 1768.32  4808.3 1769.24  4908.8 1769.79
    4933 1767.68  4962.6 1767.49  4986.8 1763.25  4993.1 1762.85  4993.6 1762.35
  5011.3 1762.85  5023.8 1766.13  5034.5 1767.23  5070.2 1767.21  5094.4    1770
    5124 1771.17  5217.7 1770.37  5239.3 1771.58    5393 1771.15  5449.8 1773.07
#Mann= 3 ,-1 , 0
    4088     .05       0  4993.1     .05       0  5011.3     .05       0
Bank Sta=4993.1,5011.3
XS Rating Curve= 0 ,0
Exp/Cntr=0.3,0.1

Type RM Length L Ch R = 1 ,17088   ,325,325,325
BEGIN DESCRIPTION:
Mapping XS 2d7542a4
END DESCRIPTION:
XS GIS Cut Line= 4
      1580780.65       6828133.3      1580943.84       6827701.8
      1581236.42      6827046.42      1581295.44      6826865.87
#Sta/Elev= 30
  4141.2 1772.19  4189.6 1771.39  4250.4 1771.62  4280.6 1770.06    4286 1770.88
  4305.4 1769.66    4341 1770.13  4499.7 1769.18  4574.5 1767.23  4591.1 1767.98
  4620.4 1767.25  4713.2 1767.49  4736.5 1768.24  4788.4 1768.29  4825.7 1767.32
  4892.2 1767.61    4979 1765.57  5004.6 1760.44  5005.1 1759.94  5022.9 1760.44
  5031.5 1763.33  5044.7 1765.11  5077.6 1765.63  5106.6 1768.44  5135.3 1769.85
  5187.2 1769.88  5228.2 1768.53  5285.7 1770.56  5371.2 1769.65  5510.2 1771.51
#Mann= 3 ,-1 , 0
  4141.2     .05       0  5004.6     .05       0  5022.9     .05       0
Bank Sta=5004.6,5022.9
XS Rating Curve= 0 ,0
Exp/Cntr=0.3,0.1

Type RM Length L Ch R = 1 ,16763   ,186,186,186
BEGIN DESCRIPTION:
Mapping XS 345938bb
END DESCRIPTION:
XS GIS Cut Line= 3
      1581423.87      6827966.62      1581418.25      6827628.12
       1581408.3      6826852.53
#Sta/Elev= 30
  4421.3 1770.03  4479.9 1768.96  4489.9 1767.13  4499.9 1766.88  4509.9  1768.1
  4579.9 1767.36  4629.9 1764.76    4710 1765.74    4800 1765.04    4830 1765.85
    4930 1765.84    4970 1765.01    4980 1763.79    4990 1761.49  4990.8 1759.75
  4991.3 1759.25  5009.1 1759.75    5040 1764.16    5080 1764.97    5110 1768.35
    5140 1769.21    5170 1769.54    5210 1769.03    5220 1768.22    5240 1769.22
    5330 1770.66    5360 1769.09    5404 1769.01    5430 1771.04  5535.5 1771.58
#Mann= 3 ,-1 , 0
  4421.3     .05       0  4990.8     .05       0  5009.1     .05       0
Bank Sta=4990.8,5009.1
XS Rating Curve= 0 ,0
Exp/Cntr=0.3,0.1

Type RM Length L Ch R = 1 ,16577   ,121,121,121
BEGIN DESCRIPTION:
Mapping XS b433ecdf
END DESCRIPTION:
XS GIS Cut Line= 3
      1581528.04      6827956.23       1581604.3       6827505.1
      1581585.22      6826752.28
#Sta/Elev= 30
  4425.2 1769.61  4474.1 1768.16  4493.1 1766.29  4504.5  1767.5  4553.6 1767.63
  4626.2 1764.57  4656.7 1764.11  4717.5 1765.57  4788.5 1765.52  4800.3 1764.79
  4839.2 1766.45  4899.8 1766.03  4959.9  1763.8  4979.9 1763.94  4999.9 1759.87
  5000.7  1759.1  5001.2  1758.6    5019  1759.1  5048.7  1763.8  5079.9 1763.97
  5099.9 1766.41  5129.9 1767.94  5199.9    1768  5229.9 1766.51  5239.9 1767.77
  5253.9 1768.07  5351.9 1768.91    5400 1768.43    5440 1769.86  5635.8 1771.36
#Mann= 5 ,-1 , 0
  4425.2     .05       0  5000.7     .05       0    5019     .05       0
  5253.9    .075       0  5351.9     .05       0
Bank Sta=5000.7,5019
XS Rating Curve= 0 ,0
Exp/Cntr=0.3,0.1

Type RM Length L Ch R = 1 ,16456   ,253,253,253
BEGIN DESCRIPTION:
Mapping XS 54a15205
END DESCRIPTION:
XS GIS Cut Line= 3
      1581750.13       6827616.2      1581724.09      6827480.79
      1581711.98      6826911.31
#Sta/Elev= 30
  4769.1 1765.34  4777.4 1764.92  4797.8 1765.25    4808 1765.83  4869.1 1766.16
  4899.6 1766.06  4959.8  1765.2  4969.8 1764.54  4979.8 1762.83  4989.8 1757.51
  4990.5 1756.24    4991 1755.74  5008.5 1755.74    5009 1756.24  5029.8 1756.46
  5039.8 1763.33  5049.8 1764.77  5059.8 1765.16  5109.8 1765.14  5149.8 1765.59
  5179.8 1765.32  5209.8  1765.5  5249.9 1766.09  5279.9 1767.06  5348.5 1767.74
  5359.9 1768.33  5369.9 1768.05  5389.9 1769.23  5452.6 1769.62  5476.6 1770.46
#Mann= 5 ,-1 , 0
  4769.1     .05       0  4990.5     .03       0    5009     .05       0
  5348.5    .075       0  5452.6     .05       0
Bank Sta=4990.5,5009
XS Rating Curve= 0 ,0
Exp/Cntr=0.3,0.1

Type RM Length L Ch R = 1 ,16203   ,413,413,413
BEGIN DESCRIPTION:
Mapping XS d0d6a131
END DESCRIPTION:
XS GIS Cut Line= 2
      1581977.57      6827617.94      1581970.62      6826848.87
#Sta/Elev= 30
  4769.7  1766.5  4829.6 1765.92  4879.6  1766.1  4909.6 1765.73  4919.6  1766.1
  4949.6 1764.88  4959.6 1763.42  4969.6  1761.1  4979.6 1759.68  4980.4 1756.24
  4980.9 1755.74  4998.4 1755.74  4998.9 1756.24  5039.6 1756.24  5049.6 1759.77
  5059.6 1762.14  5069.7 1762.65  5099.7  1763.1  5129.7 1764.44  5159.7 1764.91
  5169.7 1765.37  5249.7 1765.35  5269.7 1765.93  5299.7 1766.32  5349.7 1767.72
  5419.7 1768.47  5449.7 1767.77  5469.7 1768.44  5489.7 1768.16  5538.8 1769.34
#Mann= 3 ,-1 , 0
  4769.7     .05       0  4980.4     .05       0  4998.9     .05       0
Bank Sta=4980.4,4998.9
XS Rating Curve= 0 ,0
Exp/Cntr=0.3,0.1

Type RM Length L Ch R = 1 ,15790   ,266,266,266
BEGIN DESCRIPTION:
Mapping XS 2efc6007
END DESCRIPTION:
XS GIS Cut Line= 4
      1581921.97      6827666.57      1582262.29      6827569.34
      1582757.08      6827097.11      1582832.87      6826931.76
#Sta/Elev= 30
  4522.5 1766.17  4572.2    1766    4606 1763.84  4611.2 1764.17  4619.3 1760.66
  4629.7 1757.19  4630.5 1756.24    4631 1755.74  4648.5 1755.74    4649 1756.24
  5402.8 1756.24  5409.7 1757.08    5417 1756.32  5423.9 1758.53  5445.3 1758.98
  5452.2 1759.82  5459.4 1759.56  5466.3  1760.5  5473.6 1760.21  5480.5 1761.06
    5516 1762.65  5522.9 1763.81  5537.1 1763.91    5544 1765.12  5551.3    1765
  5556.1 1766.33  5562.7 1766.33  5566.2 1767.41  5680.4 1770.48  5742.3 1770.68
#Mann= 3 ,-1 , 0
  4522.5     .05       0  4630.5     .03       0    4649     .05       0
Bank Sta=4630.5,4649
XS Rating Curve= 0 ,0
Exp/Cntr=0.3,0.1

Type RM Length L Ch R = 1 ,15524   ,72,72,72
BEGIN DESCRIPTION:
Mapping XS 87e514bf
END DESCRIPTION:
XS GIS Cut Line= 5
      1581923.76      6827689.13      1582133.82      6827671.77
      1582706.73      6827671.77      1583106.04      6827656.14
      1583467.12      6827617.95
#Sta/Elev= 30
  4383.8 1765.73  4415.1 1765.95  4459.2 1764.05  4515.5 1757.36    4516 1756.24
  4516.5 1755.74  4535.1 1756.24  5055.8 1756.24  5105.8 1761.09  5145.8 1761.34
  5155.8 1762.39  5164.1 1765.27  5195.8 1766.73  5245.8 1765.75  5275.8 1762.66
  5295.9 1762.06  5396.3 1764.08  5415.9 1761.13    5426 1761.11    5436 1763.58
    5516 1766.38    5546 1765.24  5594.1 1761.26  5686.7 1765.61  5696.9 1764.96
  5706.8 1762.04  5777.2 1763.54  5797.3 1762.43  5867.7 1763.15  5930.2 1767.77
#Mann= 3 ,-1 , 0
  4383.8     .05       0    4516     .03       0  4535.1     .05       0
Bank Sta=4516,4535.1
XS Rating Curve= 0 ,0
Exp/Cntr=0.3,0.1

Type RM Length L Ch R = 1 ,15452   ,219,219,219
BEGIN DESCRIPTION:
Mapping XS faffaadd
END DESCRIPTION:
XS GIS Cut Line= 4
      1581929.83      6827712.71      1582296.14      6827735.28
      1582780.52      6827714.45      1583478.41       6827639.8
#Sta/Elev= 30
  4338.8 1765.26  4404.1 1763.68  4744.7  1764.1  4764.7 1763.22  4814.8 1757.06
  4874.8 1757.45  4875.3 1755.53  4875.8 1755.03  4894.4 1755.53  4914.9 1756.64
  4990.7 1755.86    5045 1756.92    5115 1760.47  5207.2 1761.35  5299.5 1760.58
    5346 1762.36  5376.2 1760.94  5391.8 1763.57  5426.4 1765.32  5496.8 1765.11
  5537.1 1761.41  5547.1 1761.44  5567.2 1765.97  5576.3 1766.11  5597.4 1764.71
  5637.6 1766.12  5738.2 1765.43  5808.6 1763.15  5848.8 1766.69  5892.5 1767.91
#Mann= 3 ,-1 , 0
  4338.8     .05       0  4875.3     .03       0  4894.4     .05       0
Bank Sta=4875.3,4894.4
XS Rating Curve= 0 ,0
Exp/Cntr=0.3,0.1

Type RM Length L Ch R = 1 ,15233   ,319,319,319
BEGIN DESCRIPTION:
Mapping XS 4510d749
END DESCRIPTION:
XS GIS Cut Line= 4
      1582082.57      6828280.43      1582462.81      6828103.34
       1582895.1      6827757.85      1583499.23      6827646.75
#Sta/Elev= 30
  4221.4 1765.77  4456.7 1764.54  4599.5 1761.62    4753 1762.21  4796.2 1760.64
  4802.6 1762.05  4831.4 1762.19  4845.9 1761.04  4860.3 1757.58  4874.1 1756.29
  4965.9 1755.79  4970.6 1754.89  4971.1 1754.39    4990 1754.89  5009.1 1756.16
  5052.4 1755.38  5079.6 1758.59  5116.4 1758.83  5143.6 1760.84  5273.4 1760.97
  5389.7  1763.4  5437.6 1761.29  5458.5 1762.17  5478.8 1765.35  5500.9 1766.15
  5692.4 1764.72  5743.2 1766.45  5771.3 1766.03  5776.4 1767.44  5808.5 1768.33
#Mann= 3 ,-1 , 0
  4221.4     .05       0  4970.6     .03       0    4990     .05       0
Bank Sta=4970.6,4990
XS Rating Curve= 0 ,0
Exp/Cntr=0.3,0.1

Type RM Length L Ch R = 1 ,14914   ,162,162,162
BEGIN DESCRIPTION:
Mapping XS 92158b0f
END DESCRIPTION:
XS GIS Cut Line= 4
      1582495.77      6828671.08      1583053.09      6827969.65
       1583395.1      6827704.03      1583511.55      6827668.07
#Sta/Elev= 30
  4262.4 1766.28  4285.4 1765.31  4299.8  1766.1  4306.2 1764.41  4320.6 1764.01
  4363.9 1764.32  4384.7 1766.35  4413.5 1766.65  4538.2 1765.51    4585 1763.47
  4698.7 1763.72  4748.4 1762.11  4769.2 1763.65  4882.9 1762.13  4897.3 1761.69
  4926.2 1755.72  5001.4 1754.42  5001.9 1753.92  5020.8 1754.42  5096.5 1754.94
  5118.4  1758.8  5156.1 1760.56  5232.3  1761.5    5417  1760.3  5466.7  1762.6
  5612.2 1765.06  5628.3 1763.73  5666.2 1763.84  5685.4 1764.75  5713.2  1769.7
#Mann= 4 ,-1 , 0
  4262.4      .1       0  4538.2     .05       0  5001.4     .03       0
  5020.8     .05       0
Bank Sta=5001.4,5020.8
XS Rating Curve= 0 ,0
Exp/Cntr=0.3,0.1

Type RM Length L Ch R = 1 ,14752   ,447,447,447
BEGIN DESCRIPTION:
Mapping XS 6b9aace9
END DESCRIPTION:
XS GIS Cut Line= 4
      1582579.63      6828755.79      1582972.88      6828310.45
      1583407.77      6827766.18      1583547.76      6827662.49
#Sta/Elev= 30
  4246.7 1766.43  4362.6 1766.61  4376.9 1766.16  4383.5 1765.21  4423.6 1764.26
    4688  1763.4  4880.1 1761.84    4908 1761.08  4958.6 1761.43  4985.8 1760.24
  4993.8  1758.8  5000.2  1756.3  5008.2 1754.36  5040.1 1754.27  5040.6 1753.77
    5059 1753.77  5059.5 1754.27  5072.2 1755.93  5107.4 1755.59  5221.1 1758.32
  5235.5 1760.21  5249.9 1760.69  5278.8 1760.24    5420 1760.39    5484 1760.81
  5533.1  1762.3  5570.8 1762.16    5648 1764.78  5677.2 1769.83  5711.7 1770.03
#Mann= 4 ,-1 , 0
  4246.7      .1       0  4423.6     .05       0  5040.1     .03       0
  5059.5     .05       0
Bank Sta=5040.1,5059.5
XS Rating Curve= 0 ,0
Exp/Cntr=0.3,0.1

Type RM Length L Ch R = 1 ,14305   ,308,308,308
BEGIN DESCRIPTION:
Mapping XS 3a87d4d5
END DESCRIPTION:
XS GIS Cut Line= 4
      1583204.62      6828659.44      1583446.84      6828375.56
      1583571.84      6828107.33       1583728.1      6827849.49
#Sta/Elev= 30
  4529.1 1766.22  4580.3  1765.4  4601.2 1762.48  4615.4 1762.17  4672.5 1763.63
  4820.7 1760.82  4935.8 1761.49  4958.7 1760.69    4976 1756.47  5011.2 1754.29
  5011.7 1753.79  5030.7 1754.29  5055.7 1755.23    5073 1760.86  5101.4 1763.19
  5186.4  1765.7  5235.8 1763.86  5272.6 1764.15  5288.1 1765.87    5294 1764.94
  5309.5 1767.15  5315.3 1766.08    5325 1767.43  5330.8 1765.89  5346.3  1768.3
  5354.9 1767.46  5367.6 1769.02  5423.2 1770.52  5467.5 1770.91  5499.7 1770.86
#Mann= 6 ,-1 , 0
  4529.1     .05       0  5011.2     .03       0  5030.7     .05       0
  5354.9    .075       0  5423.2     .05       0  5467.5    .075       0
Bank Sta=5011.2,5030.7
XS Rating Curve= 0 ,0
Exp/Cntr=0.3,0.1

Type RM Length L Ch R = 1 ,13997   ,489,489,489
BEGIN DESCRIPTION:
Mapping XS b5635808
END DESCRIPTION:
XS GIS Cut Line= 4
      1583720.25      6828524.04      1583772.36      6828443.27
      1583777.57      6827940.66      1583837.45      6827766.21
#Sta/Elev= 30
  4719.2 1763.47  4734.8 1763.41  4740.7    1760  4749.9 1759.49  4755.9 1756.35
  4771.1 1755.88    4777 1754.28  4798.1 1755.53  4807.4 1755.34  4813.1  1756.3
  4830.6 1755.26  4910.6 1755.63  4950.6 1755.32  4960.6  1754.5  4980.6 1755.89
  4990.8 1753.52  4991.3 1753.02  5010.3 1753.52  5010.6 1755.09  5030.6 1754.35
  5110.6 1760.63  5170.6 1763.07  5250.6 1763.72  5300.6 1765.16  5351.7 1764.68
  5445.5 1767.29  5485.3  1766.8  5489.9 1766.68  5498.8 1768.49  5502.4 1768.49
#Mann= 4 ,-1 , 0
  4719.2     .05       0  4990.8     .03       0  5010.3     .05       0
  5485.3    .075       0
Bank Sta=4990.8,5010.3
XS Rating Curve= 0 ,0
Exp/Cntr=0.3,0.1

Type RM Length L Ch R = 1 ,13508   ,368,368,368
BEGIN DESCRIPTION:
Mapping XS 30b351c3
END DESCRIPTION:
XS GIS Cut Line= 3
      1583722.88       6828651.6      1584274.96      6828550.04
      1584319.23        6828524.
#Sta/Elev= 30
  4662.3 1762.64  4674.6 1761.57  4684.8 1757.99    4695  1755.6    4710  1754.7
  4715.3 1756.12  4776.3 1758.23  4821.2 1758.28  4837.3  1757.7  4867.8  1757.6
  4908.5 1758.01  4932.4 1756.72  4959.3 1753.13  4969.5 1753.51  4975.7 1751.73
  4976.2 1751.23  4994.7 1751.23  4995.2 1751.73    5000 1752.74  5020.3 1753.38
  5043.6 1753.08    5061 1755.66  5111.9 1758.39  5142.3 1758.84  5172.8 1761.47
  5202.8 1760.84  5207.9 1761.29  5233.5 1760.61  5239.3 1760.95    5275 1760.63
#Mann= 4 ,-1 , 0
  4662.3     .05       0  4975.7     .03       0  4995.2     .05       0
  5111.9      .1       0
Bank Sta=4975.7,4995.2
XS Rating Curve= 0 ,0
Exp/Cntr=0.3,0.1

Type RM Length L Ch R = 1 ,13140   ,391,391,391
BEGIN DESCRIPTION:
Mapping XS 487a3c04
END DESCRIPTION:
XS GIS Cut Line= 3
      1583811.44      6829141.16      1584225.48      6828706.29
      1584316.61      6828617.77
#Sta/Elev= 30
    4649 1761.78  4660.8 1761.53  4667.7 1758.72    4675 1757.93  4681.9 1756.12
  4696.1 1755.12  4703.3 1755.32  4710.2 1757.26  4762.3 1756.22  4861.1 1756.26
  4922.5 1756.01  4943.6 1756.78  4950.8 1755.64  4955.3 1750.38  4955.8 1749.88
  4974.8 1750.38  4993.3 1752.93  5007.5 1752.52  5042.7  1754.1  5049.9 1753.67
  5092.4 1756.56  5163.2 1757.37  5212.5 1756.65  5251.8 1757.81  5262.1 1758.63
  5269.1 1760.49  5283.3 1761.62    5294 1761.45  5299.3 1761.34  5376.5 1760.46
#Mann= 7 ,-1 , 0
    4649     .05       0  4762.3    .075       0  4861.1     .05       0
  4955.3     .03       0  4974.8     .05       0    5294    .075       0
  5299.3      .1       0
Bank Sta=4955.3,4974.8
XS Rating Curve= 0 ,0
Exp/Cntr=0.3,0.1

Type RM Length L Ch R = 1 ,12749   ,285,285,285
BEGIN DESCRIPTION:
Mapping XS 66fb42b1
END DESCRIPTION:
XS GIS Cut Line= 4
      1583902.58      6829396.39        1584301.      6829219.31
      1584535.38      6828734.93      1584590.03      6828456.45
#Sta/Elev= 30
  4362.2 1761.47  4393.7 1757.44  4422.4 1758.94  4544.2  1756.7  4657.5 1756.38
  4671.4 1757.04  4717.9 1756.17  4780.7 1756.53  4793.1 1754.76  4817.6 1754.51
  4845.7 1756.27  4907.9 1755.18  4958.7 1756.23  4975.7 1753.69  4981.3 1753.93
  4994.1 1750.47  4994.6 1749.97  5013.7 1750.47    5049 1751.89  5066.1 1755.95
  5106.4 1755.56  5177.4 1755.64    5244 1757.78  5303.1 1758.03  5320.1 1756.67
  5336.3 1756.67  5384.1 1758.46  5439.3 1759.13  5577.8 1758.96  5620.1 1760.11
#Mann= 6 ,-1 , 0
  4362.2    .075       0  4657.5     .05       0  4994.1     .03       0
  5013.7     .05       0  5106.4    .075       0  5439.3      .1       0
Bank Sta=4994.1,5013.7
XS Rating Curve= 0 ,0
Exp/Cntr=0.3,0.1

Type RM Length L Ch R = 1 ,12464   ,330,330,330
BEGIN DESCRIPTION:
Mapping XS 2e394a8a
END DESCRIPTION:
XS GIS Cut Line= 3
      1584428.61      6829823.46      1584717.67      6828846.91
      1584746.32      6828576.05
#Sta/Elev= 30
  4335.1 1759.21  4495.7 1757.65  4601.5 1757.72  4674.5 1755.86  4747.5 1756.37
  4841.4 1755.39  4887.1 1755.93  4939.7 1754.97  4956.1 1755.43  4971.7 1753.41
  4977.6 1749.61  4978.1 1749.11  4996.7 1749.11  4997.2 1749.61  5018.7  1755.2
  5021.9 1755.17  5158.3 1755.41  5188.2 1755.43    5196 1756.05  5206.4 1755.04
  5216.2 1754.96  5300.3 1756.62  5353.5 1756.28  5376.6  1756.9  5382.7 1757.85
  5493.2 1756.82  5503.3 1756.96  5523.4 1758.93  5540.2 1759.19  5625.9 1759.42
#Mann= 9 ,-1 , 0
  4335.1     .05       0  4495.7    .075       0  4887.1     .05       0
  4977.6     .03       0  4997.2     .05       0  5021.9    .075       0
  5158.3      .1       0  5382.7    .075       0  5540.2      .1       0
Bank Sta=4977.6,4997.2
XS Rating Curve= 0 ,0
Exp/Cntr=0.3,0.1

Type RM Length L Ch R = 1 ,12134   ,215,215,215
BEGIN DESCRIPTION:
Mapping XS c788af26
END DESCRIPTION:
XS GIS Cut Line= 3
      1584933.82      6829922.42      1584933.82      6829240.14
       1584923.4      6828703.72
#Sta/Elev= 30
  4215.8 1759.76  4345.5 1758.45  4369.5 1758.33  4460.2 1756.95  4510.2 1755.37
  4550.2 1756.08  4582.2 1755.97  4640.2 1756.09  4650.2 1755.29  4670.2 1756.36
  4730.2 1755.88  4759.1 1756.33  4800.2  1756.2  4840.2 1754.99  4880.2 1755.38
  4896.6  1754.7  4970.2 1754.07  4980.2 1753.63  4990.2 1751.65  4990.4 1749.26
  4990.9 1748.76  5009.6 1748.76  5010.1 1749.26  5010.2 1749.71  5030.2 1751.35
  5040.2  1753.7  5050.2 1754.44  5212.2 1755.66  5343.4 1756.25  5434.6 1756.62
#Mann= 9 ,-1 , 0
  4215.8    .075       0  4345.5      .1       0  4369.5    .075       0
  4582.2      .1       0  4759.1    .075       0  4990.4     .07       0
  5010.1    .075       0  5212.2      .1       0  5343.4    .075       0
Bank Sta=4990.4,5010.1
XS Rating Curve= 0 ,0
Exp/Cntr=0.3,0.1

Type RM Length L Ch R = 1 ,11919   ,465,465,465
BEGIN DESCRIPTION:
Mapping XS c34731e7
END DESCRIPTION:
XS GIS Cut Line= 2
      1585147.36       6829745.4      1585144.75       6828594.3
#Sta/Elev= 30
  4393.5 1756.54  4558.2 1755.48  4620.9  1753.7  4656.1 1754.04  4690.9  1754.7
    4754 1753.53  4830.9 1753.75  4930.9 1752.95  4970.9 1751.89  4980.9 1748.88
    4991 1748.36  4991.5 1747.86  5010.2 1747.86  5010.7 1748.36  5010.9 1749.25
  5040.9 1751.37  5060.9 1752.09  5080.9 1755.17  5100.9 1756.14  5180.9 1755.83
  5210.9 1756.63  5240.9 1756.57  5300.9 1755.39  5330.9 1755.44  5380.9 1756.98
  5416.1 1757.07  5450.9 1757.04  5460.9 1757.73  5520.9 1758.89  5544.6 1758.73
#Mann= 7 ,-1 , 0
  4393.5      .1       0  4558.2     .05       0  4656.1      .1       0
    4754     .05       0    4991     .07       0  5010.7     .05       0
  5416.1      .1       0
Bank Sta=4991,5010.7
XS Rating Curve= 0 ,0
Exp/Cntr=0.3,0.1

Type RM Length L Ch R = 1 ,11454   ,362,362,362
BEGIN DESCRIPTION:
Mapping XS ba0a7ea9
END DESCRIPTION:
XS GIS Cut Line= 2
      1585511.94      6829758.34      1585530.17       6828714.1
#Sta/Elev= 30
  4628.2 1755.66  4668.5  1755.8  4748.6 1754.99  4788.6 1755.21  4848.6 1753.62
  4878.6 1753.48  4948.6 1754.29  4968.6 1753.62  5018.6 1748.84  5018.8 1748.42
  5019.3 1747.92    5038 1747.92  5038.5 1748.42  5038.6 1750.24  5048.6 1752.36
  5058.6 1752.03  5086.8 1752.65  5188.6 1752.61  5248.6 1753.64  5278.6 1753.36
  5298.6 1754.62  5338.6  1754.2  5378.7 1754.58  5408.7 1753.79  5512.2 1754.32
  5548.7 1753.58  5558.7 1753.97  5578.7  1753.7  5608.7  1755.4  5672.6 1756.33
#Mann= 4 ,-1 , 0
  4628.2     .05       0  5018.8     .03       0  5038.5     .05       0
  5512.2    .075       0
Bank Sta=5018.8,5038.5
XS Rating Curve= 0 ,0
Exp/Cntr=0.3,0.1

Type RM Length L Ch R = 1 ,11092   ,592,592,592
BEGIN DESCRIPTION:
Mapping XS 43acea3a
END DESCRIPTION:
XS GIS Cut Line= 4
      1585881.73      6829875.52      1585876.52      6829372.95
      1585707.25      6828945.87      1585730.57      6828601.26
#Sta/Elev= 30
  4352.5 1760.36  4431.5 1758.91    4480 1757.66    4510 1753.67  4529.5 1753.48
    4540  1752.9    4560 1753.79    4640 1754.46    4820 1752.44  4881.9 1752.64
  4946.5 1750.84    4953 1750.15  4958.4 1748.59  5002.6 1748.37  5003.1 1747.87
  5021.9 1747.87  5022.4 1748.37  5031.4 1751.21  5097.1 1751.97  5236.9 1751.41
  5269.2 1751.75  5290.7 1753.48  5310.8 1753.92  5411.3 1753.98  5422.6 1752.97
  5462.7 1752.92  5512.8 1755.75  5613.1 1756.64  5633.1 1757.82  5659.9 1758.24
#Mann= 6 ,-1 , 0
  4352.5     .05       0  4431.5    .075       0  4529.5     .05       0
  5002.6     .03       0  5022.4     .05       0  5411.3    .075       0
Bank Sta=5002.6,5022.4
XS Rating Curve= 0 ,0
Exp/Cntr=0.3,0.1

Type RM Length L Ch R = 1 ,10500   ,446,446,446
BEGIN DESCRIPTION:
Mapping XS c1de6199
END DESCRIPTION:
XS GIS Cut Line= 4
      1585963.77      6829838.65      1586028.87      6829492.31
      1586375.22      6829132.94      1586388.24      6828635.52
#Sta/Elev= 30
  4393.6 1761.28    4434 1760.17  4506.2  1757.8  4526.5 1754.54  4533.1 1754.55
  4557.1 1753.68  4586.1 1754.82  4689.3 1754.34  4788.8 1752.04  4802.9  1750.5
  4809.9 1748.39  4884.8 1748.34  4885.3 1747.84  4904.7 1748.34  5092.9 1748.39
  5099.8 1751.99    5107 1751.36    5114 1752.75  5133.9 1752.91  5142.3 1753.89
  5149.5 1752.58  5156.4 1754.15  5163.6 1752.86  5170.6 1754.14  5191.9  1752.2
  5234.4 1751.16  5370.1 1750.31  5547.3 1753.39  5640.2 1755.25  5742.7  1755.9
#Mann= 6 ,-1 , 0
  4393.6     .05       0    4434    .075       0  4533.1     .05       0
  4884.8     .03       0  4904.7     .05       0  5547.3    .075       0
Bank Sta=4884.8,4904.7
XS Rating Curve= 0 ,0
Exp/Cntr=0.3,0.1

Type RM Length L Ch R = 1 ,10054   ,191,191,191
BEGIN DESCRIPTION:
Mapping XS d9c1a917
END DESCRIPTION:
XS GIS Cut Line= 4
      1586591.37      6829992.35      1586586.16      6829416.79
      1586437.72      6829101.69      1586471.46      6828611.24
#Sta/Elev= 30
  4266.5 1752.85  4380.9 1751.69  4480.9 1751.81  4507.1 1750.76  4570.9 1748.96
  4590.9 1750.19  4610.9 1750.35    4639 1752.24  4770.9 1751.25  4879.7  1754.5
    4896 1748.37  4938.1 1748.32  4938.6 1747.82  4957.5 1747.82    4958 1748.32
  5073.1 1748.39  5083.9 1749.37  5090.3 1750.86    5106 1752.88  5118.6 1753.65
  5141.4 1752.86  5158.7 1751.41  5226.4 1750.26  5294.3 1750.71  5324.4 1752.15
  5384.5 1751.54  5459.9  1752.9  5494.8 1753.22  5534.9 1754.73    5682 1755.12
#Mann= 6 ,-1 , 0
  4266.5      .1       0  4507.1    .075       0    4639     .05       0
  4938.1     .03       0    4958     .05       0  5459.9    .075       0
Bank Sta=4938.1,4958
XS Rating Curve= 0 ,0
Exp/Cntr=0.3,0.1

Type RM Length L Ch R = 1 ,9863    ,185,185,185
BEGIN DESCRIPTION:
Mapping XS 193d7726
END DESCRIPTION:
XS GIS Cut Line= 4
      1586687.72      6830013.12      1586703.35      6829263.14
      1586656.47      6829127.73      1586601.78      6828586.02
#Sta/Elev= 30
  4169.8  1752.3  4183.4 1752.49  4234.9 1752.48  4294.9 1751.04    4405  1751.7
  4436.9 1750.06    4495 1748.61    4515 1750.18  4560.2 1750.12    4625 1751.76
    4675 1750.81    4715 1753.06  4754.6 1753.95  4765.1 1752.08  4795.1 1750.09
  4905.1 1749.93  4919.9 1750.39  4930.4 1751.97  4946.5 1751.77  4961.6 1748.44
  5021.2  1748.3  5021.7  1747.8  5041.3  1748.3  5049.8 1749.02  5113.2 1748.41
    5128 1750.12    5355 1751.55  5444.9 1753.68  5500.6 1753.74  5607.7 1753.46
#Mann= 8 ,-1 , 0
  4169.8    .075       0  4183.4      .1       0  4436.9    .075       0
  4560.2     .05       0  5021.2     .03       0  5041.3     .05       0
    5355    .075       0  5500.6     .05       0
Bank Sta=5021.2,5041.3
XS Rating Curve= 0 ,0
Exp/Cntr=0.3,0.1

Type RM Length L Ch R = 1 ,9678    ,581,581,581
BEGIN DESCRIPTION:
Mapping XS 57e10cbd
END DESCRIPTION:
XS GIS Cut Line= 2
      1586856.99      6829994.89      1586836.16      6828494.94
#Sta/Elev= 30
  4245.3 1752.06  4262.2 1752.31  4292.2 1750.65  4302.5 1750.77  4362.2 1750.04
  4452.2 1750.61  4502.9 1748.93  4552.2 1748.19  4613.2 1750.11  4842.3 1748.94
  4902.3 1751.28  4962.3 1747.07  4972.3 1745.37  4982.2  1741.5  4982.7    1741
  5002.3  1741.5  5012.3 1741.94  5022.3 1744.88  5032.3 1746.71  5062.3 1750.24
  5122.3 1751.75  5182.3 1751.07  5362.3 1752.68  5382.3 1752.59  5402.3 1751.09
    5495 1751.83  5623.7  1752.1  5672.3 1753.48  5692.3 1752.67  5745.4 1753.88
#Mann= 8 ,-1 , 0
  4245.3    .075       0  4302.5      .1       0  4502.9    .075       0
  4613.2     .05       0  4982.2     .03       0  5002.3     .05       0
    5495      .1       0  5623.7     .05       0
Bank Sta=4982.2,5002.3
XS Rating Curve= 0 ,0
Exp/Cntr=0.3,0.1

Type RM Length L Ch R = 1 ,9097    ,623,623,623
BEGIN DESCRIPTION:
Mapping XS 61db16a8
END DESCRIPTION:
XS GIS Cut Line= 2
      1587370.01      6829864.67      1587393.45      6828614.69
#Sta/Elev= 30
    4422 1750.31  4508.7  1750.1  4558.7  1748.3  4578.7 1746.81  4591.8 1746.88
  4628.7 1746.43  4878.8 1748.06  4938.8 1746.67  4948.8 1746.21  4954.2 1745.56
  4959.2 1744.29  4978.8 1744.52  4988.8 1743.94  5008.7  1740.5  5009.2    1740
  5028.3    1740  5028.8  1740.5  5038.8 1743.98  5048.8 1745.95  5078.8 1746.75
  5198.8 1747.26  5288.8 1746.63  5338.8 1747.64  5378.8 1749.28  5469.2 1750.73
  5498.9 1751.49  5518.9 1750.59  5588.9 1752.12  5618.9 1753.24  5672.2 1753.12
#Mann= 5 ,-1 , 0
    4422      .1       0  4591.8     .05       0  5008.7     .04       0
  5028.8     .05       0  5469.2      .1       0
Bank Sta=5008.7,5028.8
XS Rating Curve= 0 ,0
Exp/Cntr=0.3,0.1

Type RM Length L Ch R = 1 ,8474    ,463,463,463
BEGIN DESCRIPTION:
Mapping XS 420ad8fb
END DESCRIPTION:
XS GIS Cut Line= 3
       1587502.8      6829817.86      1587950.74      6829408.98
      1588122.25       6828611.2
#Sta/Elev= 30
  4270.1 1748.35  4385.1  1746.7  4420.4 1746.69  4427.2 1745.37  4441.4 1745.04
  4476.5 1745.86  4504.9 1745.14  4569.1 1745.76  4646.8 1745.08  4667.7 1746.02
  4760.3 1744.64  4898.1 1745.41  5000.3 1742.85  5000.4 1740.56  5000.9 1740.06
  5020.7 1740.56  5051.5 1741.98    5060 1743.48  5065.1 1742.93  5082.2  1744.1
  5123.1 1742.93  5133.3  1744.2  5143.5 1744.08  5153.6 1742.45  5158.7 1742.53
    5164  1743.9  5184.5 1744.89  5368.6 1745.75  5409.5 1748.89  5692.6 1754.55
#Mann= 4 ,-1 , 0
  4270.1      .1       0  4385.1     .05       0  5000.4     .05       0
  5020.7     .05       0
Bank Sta=5000.4,5020.7
XS Rating Curve= 0 ,0
Exp/Cntr=0.3,0.1

Type RM Length L Ch R = 1 ,8011    ,373,373,373
BEGIN DESCRIPTION:
Mapping XS 5e2f491a
END DESCRIPTION:
XS GIS Cut Line= 3
      1587521.04      6829828.25      1588190.33      6829614.71
      1588744.49      6829242.66
#Sta/Elev= 30
  4159.1 1748.81  4236.9 1748.23  4415.2 1746.37  4504.9  1746.5  4520.1 1747.25
  4562.1 1746.35  4574.5 1745.46  4665.9 1745.25    4698 1745.73  4709.1 1744.91
  4730.1 1744.57  4772.9 1745.18  4832.1 1743.84    4856 1744.29  4897.4 1742.92
  4915.8 1743.73    4971 1742.48  4981.8 1741.39  4982.3 1740.89  5001.7 1740.89
  5002.2 1741.39    5022 1741.55    5028 1742.24    5079 1742.64    5094 1743.48
    5121 1746.22    5136 1745.77  5331.1 1750.79  5511.1 1752.71  5529.1 1752.45
#Mann= 6 ,-1 , 0
  4159.1      .1       0  4236.9     .05       0  4897.4     .12       0
  4915.8     .05       0  4981.8     .05       0  5002.2     .05       0
Bank Sta=4981.8,5002.2
XS Rating Curve= 0 ,0
Exp/Cntr=0.3,0.1

Type RM Length L Ch R = 1 ,7638    ,369,369,369
BEGIN DESCRIPTION:
Mapping XS 6aa75506
END DESCRIPTION:
XS GIS Cut Line= 4
      1587609.62      6829901.16      1588278.87      6829849.08
      1588583.56      6829789.19      1588836.13      6829497.55
#Sta/Elev= 30
    4120 1749.54  4366.1 1746.34  4426.3 1746.55  4436.3  1745.1  4466.4  1744.2
  4526.6 1743.98  4546.7 1745.03  4566.7 1744.11  4596.8 1744.53  4611.9 1743.63
  4616.9 1744.67  4717.2 1745.03  4848.5 1744.05  4889.2 1744.61  4925.7 1742.76
  4940.2 1743.06  4977.1 1740.42  4991.2 1737.35  4991.7 1736.85  5011.1 1736.85
  5011.6 1737.35  5028.5 1741.64  5033.6 1741.02  5038.1 1741.84  5052.3 1743.34
  5067.5 1743.76  5093.1 1744.18  5117.4 1743.73  5202.9 1744.98  5487.6  1747.3
#Mann= 5 ,-1 , 0
    4120     .05       0  4991.2     .04       0  5011.6     .05       0
  5038.1     .12       0  5067.5     .05       0
Bank Sta=4991.2,5011.6
XS Rating Curve= 0 ,0
Exp/Cntr=0.3,0.1

Type RM Length L Ch R = 1 ,7269    ,737,737,737
BEGIN DESCRIPTION:
Mapping XS 62c1203c
END DESCRIPTION:
XS GIS Cut Line= 4
      1587656.43      6830114.71      1588370.01      6830122.52
      1588613.89      6830110.68      1589249.41      6829794.77
#Sta/Elev= 30
    4052 1748.75  4056.2 1748.73  4080.6 1748.59  4130.6 1746.26  4150.6 1746.62
  4220.6 1745.05  4330.6 1743.77  4550.6 1742.88  4640.6 1741.06  4760.6 1740.85
  4947.2 1742.34  4958.9 1741.42  4963.9 1740.06  4970.7 1734.29  4971.2 1733.79
  4991.1 1734.29  5000.9 1739.41  5007.8  1741.9  5037.7 1742.93  5273.8 1740.49
    5369 1740.59  5408.2 1739.75  5525.8 1741.44  5548.2 1742.38  5558.2  1741.7
  5580.6 1742.36    5593 1741.52  5637.8 1741.58    5705 1742.54  5719.5 1743.44
#Mann= 6 ,-1 , 0
    4052    .075       0  4056.2     .05       0  4947.2     .12       0
  4970.7     .06       0  4991.1     .12       0  5037.7     .05       0
Bank Sta=4970.7,4991.1
XS Rating Curve= 0 ,0
Exp/Cntr=0.3,0.1

Type RM Length L Ch R = 1 ,6532    ,495,495,495
BEGIN DESCRIPTION:
Mapping XS 10f6f6a5
END DESCRIPTION:
XS GIS Cut Line= 4
      1587573.18      6830528.77      1588093.97      6830507.94
      1588458.56      6830578.25      1588646.05      6830552.21
#Sta/Elev= 30
  4275.9 1748.91  4397.8 1748.37  4437.8 1746.02  4527.9 1744.54  4547.9 1743.62
    4598 1742.68  4800.2 1741.98  4875.6 1740.35  4920.4 1741.13  4940.7 1740.59
  4950.9 1739.48  4973.8 1738.91  4984.4 1739.35  5001.8 1734.94  5002.3 1734.44
  5021.7 1734.44  5022.2 1734.94  5031.2 1740.62  5036.3    1741  5052.8 1740.46
  5062.9 1739.32  5091.4 1739.31  5103.7 1739.66  5124.1 1739.09    5140 1739.82
  5235.5 1740.24    5286 1742.52  5326.4 1742.99  5346.5 1744.15  5357.7 1743.96
#Mann= 5 ,-1 , 0
  4275.9     .05       0  4973.8     .12       0  5001.8     .07       0
  5022.2     .12       0  5091.4     .05       0
Bank Sta=5001.8,5022.2
XS Rating Curve= 0 ,0
Exp/Cntr=0.3,0.1

Type RM Length L Ch R = 1 ,6037    ,645,645,645
BEGIN DESCRIPTION:
Mapping XS 61606178
END DESCRIPTION:
XS GIS Cut Line= 4
      1587476.79      6831078.25      1587940.33      6831052.21
      1588653.87      6830742.31      1588768.45      6830643.35
#Sta/Elev= 30
  4323.9 1746.16  4402.2 1745.84  4432.3 1746.42  4512.4 1745.37  4542.5 1746.42
  4591.6 1745.19  4702.7 1745.09  4804.2 1743.71  4914.9 1741.16  4967.7 1740.28
  4978.6 1738.39  4980.8 1734.12  4981.3 1733.62  5000.7 1733.62  5001.2 1734.12
    5009 1737.15  5014.4 1738.36    5044 1739.92  5151.2 1739.53    5273 1739.54
  5305.7 1738.94  5327.5 1739.82  5341.1 1739.17    5382  1739.1  5411.5 1739.87
  5487.3 1739.23    5620 1740.91  5655.2  1741.7    5676 1742.91  5717.5 1742.79
#Mann= 5 ,-1 , 0
  4323.9     .05       0  4914.9     .12       0  4980.8     .07       0
  5001.2     .12       0  5151.2     .05       0
Bank Sta=4980.8,5001.2
XS Rating Curve= 0 ,0
Exp/Cntr=0.3,0.1

Type RM Length L Ch R = 1 ,5392    ,333,333,333
BEGIN DESCRIPTION:
Mapping XS 96472b9e
END DESCRIPTION:
XS GIS Cut Line= 3
      1587922.11      6831289.19      1588789.28      6831281.37
      1589101.12      6831268.78
#Sta/Elev= 30
  4316.7 1743.99  4329.6 1743.98  4349.6 1742.76  4359.6 1742.49  4409.6 1742.01
  4519.6 1739.97  4779.6 1738.05  4919.6 1737.91  4979.6 1736.15  4989.6 1735.51
  4999.4 1733.96  4999.9 1733.46  5019.4 1733.46  5019.9 1733.96  5029.6 1735.91
  5059.6 1736.89  5089.6  1737.5  5109.6 1737.44  5119.6 1737.73  5199.6 1738.49
  5309.7 1738.58  5329.7 1739.19  5349.8 1739.45  5379.1 1738.68  5388.1 1738.49
  5393.1 1738.86  5419.8 1738.94  5439.8 1738.32  5469.9 1739.72    5496 1740.13
#Mann= 4 ,-1 , 0
  4316.7     .05       0  4999.4     .03       0  5019.9     .05       0
  5379.1    .075       0
Bank Sta=4999.4,5019.9
XS Rating Curve= 0 ,0
Exp/Cntr=0.3,0.1

Type RM Length L Ch R = 1 ,5059    ,370,370,370
BEGIN DESCRIPTION:
Mapping XS 265b04e7
END DESCRIPTION:
XS GIS Cut Line= 4
      1587893.45      6831317.83      1588448.14      6831510.54
      1588695.99      6831691.01      1588881.71      6831740.48
#Sta/Elev= 30
    4286  1743.7  4382.9 1742.46  4520.5 1739.68  4634.3 1738.74  4689.9 1737.61
  4721.7 1736.36  4742.8 1737.66  4753.4 1737.51  4758.8 1736.49  4764.1  1736.3
  4789.9  1736.1  4827.5 1736.73  4941.4 1736.64  4962.2 1736.24  4976.9 1735.34
  4983.1 1734.92  4987.5 1733.72    4988 1733.22  5007.5 1733.22    5008 1733.72
  5018.6 1734.11  5033.3 1735.38  5062.7 1736.56  5112.9 1737.55  5181.9 1737.57
  5282.3 1736.66  5300.9 1737.97  5313.3  1738.3  5363.5 1738.34    5372 1738.42
#Mann= 4 ,-1 , 0
    4286     .05       0  4987.5     .03       0    5008     .05       0
  5363.5     .12       0
Bank Sta=4987.5,5008
XS Rating Curve= 0 ,0
Exp/Cntr=0.3,0.1
