--- Cedar Creek.prj (project) ---

Proj Title=Cedar Creek Base Level Engineering
Current Plan=p01
Default Exp/Contr=0.3,0.1
English Units
Geom File=g01
Flow File=f01
Plan File=p01
BEGIN DESCRIPTION:
Cedar Creek
END DESCRIPTION:

--- Cedar Creek.p01 (plan) ---

Plan Title=Multiple Run
Short Identifier=Multiple
Geom File=g01
Flow File=f01
Subcritical Flow
K Sum by GR= 0
Std Step Tol= 0.01
Critical Tol= 0.01
Num of Std Step Trials= 20
Max Error Tol= 0.3
Flow Tol Ratio= 0.001
Split Flow NTrial= 30
Split Flow Tol= 0.02
Split Flow Ratio= 0.02
Log Output Level= 0
Friction Slope Method= 1
Unsteady Friction Slope Method= 2
Unsteady Bridges Friction Slope Method= 1
Parabolic Critical Depth
Global Vel Dist=  1 , 1 , 1
Global Log Level= 0
CheckData=True
Encroach Param= -1, 0, 0, 0
BEGIN DESCRIPTION:
Multiple Run
END DESCRIPTION:

--- Cedar Creek.f01 (steady flow) ---

Flow Title=Multiple
Number of Profiles=7
Profile Names=10-year,25-year,50-year,1pct_min,100-year,1pct_plu,500-year
River Rch & RM= Cedar Creek,Reach-1,176820
      80     103     122      89     143     197     200
River Rch & RM= Cedar Creek,Reach-1,174481
     282     395     491     378     605     833     934
River Rch & RM= Cedar Creek,Reach-1,167841
     374     533     667     518     830    1140    1300
River Rch & RM= Cedar Creek,Reach-1,165753
     456     654     822     640    1030    1410    1620
River Rch & RM= Cedar Creek,Reach-1,161046
     660     959    1220     954    1530    2100    2450
River Rch & RM= Cedar Creek,Reach-1,158156
    1050    1550    2000    1580    2540    3490    4160
River Rch & RM= Cedar Creek,Reach-1,155708
    1620    2460    3230    2610    4190    5770    7150
River Rch & RM= Cedar Creek,Reach-1,147917
    1860    2820    3690    2980    4770    6570    8090
River Rch & RM= Cedar Creek,Reach-1,136080
    1920    2900    3790    3050    4890    6730    8260
River Rch & RM= Cedar Creek,Reach-1,128767
    1930    2910    3790    3040    4870    6700    8170
River Rch & RM= Cedar Creek,Reach-1,123994
    1970    2960    3850    3080    4930    6780    8200
River Rch & RM= Cedar Creek,Reach-1,110549
    1930    2880    3720    2960    4740    6520    7810
River Rch & RM= Cedar Creek,Reach-1,93881
    2350    3520    4560    3630    5820    8000    9610
River Rch & RM= Cedar Creek,Reach-1,83077
    2350    3490    4500    3570    5720    7880    9380
River Rch & RM= Cedar Creek,Reach-1,60072
    2730    4080    5270    4190    6720    9240   11100
River Rch & RM= Cedar Creek,Reach-1,58286
    2820    4200    5420    4300    6900    9490   11300
River Rch & RM= Cedar Creek,Reach-1,47172
    4560    7070    9390    8050   12900   17800   21300
River Rch & RM= Cedar Creek,Reach-1,30534
    4530    7010    9310    7990   12800   17600   21100
River Rch & RM= Cedar Creek,Reach-1,24223
    4470    6920    9180    7880   12600   17400   20700
River Rch & RM= Cedar Creek,Reach-1,14028
    5360    8150   10700    8770   14100   19300   23200
River Rch & RM= Cedar Creek,Reach-1,7277
    5820    8750   11400    9100   14600   20100   24200
River Rch & RM= Cedar Creek,Reach-1,3473
    5870    8820   11500    9160   14700   20200   24300
Boundary for River Rch & Prof#=Cedar Creek,Reach-1,1
Up Type=0
Dn Type=3
Dn Slope=0.0001
Boundary for River Rch & Prof#=Cedar Creek,Reach-1,2
Up Type=0
Dn Type=3
Dn Slope=0.0001
Boundary for River Rch & Prof#=Cedar Creek,Reach-1,3
Up Type=0
Dn Type=3
Dn Slope=0.0001
Boundary for River Rch & Prof#=Cedar Creek,Reach-1,4
Up Type=0
Dn Type=3
Dn Slope=0.0001
Boundary for River Rch & Prof#=Cedar Creek,Reach-1,5
Up Type=0
Dn Type=3
Dn Slope=0.0001
Boundary for River Rch & Prof#=Cedar Creek,Reach-1,6
Up Type=0
Dn Type=3
Dn Slope=0.0001
Boundary for River Rch & Prof#=Cedar Creek,Reach-1,7
Up Type=0
Dn Type=3
Dn Slope=0.0001

--- Cedar Creek.g01 (geometry) ---

Geom Title=Existing Conditions

River Reach=Cedar Creek,Reach-1
Reach XY= 30
      1585105.00      6767338.00      1580509.96      6770143.11
      1579207.45      6773282.54      1574710.44      6774490.17
      1572754.01      6776807.05      1575414.01      6785745.02
      1577653.87      6787500.03      1578112.07      6791838.01
      1583199.54      6797385.55      1584597.21      6801434.57
      1583658.61      6802136.50      1586310.58      6807533.24
      1588100.03      6808135.41      1587858.54      6811536.54
      1589552.88      6812293.27      1587656.38      6823978.34
      1589955.61      6830258.61      1588062.80      6833034.58
      1588994.48      6834397.79      1587154.64      6835519.74
      1590452.64      6840843.52      1590807.34      6847032.51
      1592103.76      6847597.70      1593004.93      6853767.97
      1591258.42      6856836.78      1595547.23      6864234.59
      1594408.54      6865636.54      1596397.55      6867331.95
      1597755.00      6872188.00      1595455.00      6877338.00

Type RM Length L Ch R = 1,176820,197,197,197
BEGIN DESCRIPTION:
Cedar Creek 176470.516
END DESCRIPTION:
XS GIS Cut Line= 3
      1585034.26      6767068.23      1585089.53      6767353.63
      1585215.76      6767644.30
#Sta/Elev= 30
  4709.3 2015.83  4737.0 2014.28  4742.1 2014.49  4749.8 2013.85  4788.8 2011.71
  4793.9 2011.90  4810.9 2010.78  4840.5 2009.44  4845.6 2009.53  4872.0 2008.28
  4897.4 2008.07  4949.1 2007.11  4954.2 2007.47  4971.9 2006.76  4972.1 2006.26
  4975.6 2006.26  4975.9 2006.76  5005.7 2007.37  5029.1 2007.30  5037.5 2007.75
  5070.2 2007.65  5081.5 2008.01  5092.0 2007.77  5123.0 2008.41  5157.4 2009.47
  5175.3 2009.65  5280.0 2013.17  5298.1 2013.50  5303.5 2013.83  5316.9 2013.94
#Mann=3,-1,0
  4709.3    0.05       0  4971.9    0.05       0  4975.9    0.05       0
Bank Sta=4971.9,4975.9
Exp/Cntr=0.3,0.1

Type RM Length L Ch R = 1,176623,49,49,49
BEGIN DESCRIPTION:
Cedar Creek 176623.2
END DESCRIPTION:
XS GIS Cut Line= 3
      1584871.28      6767088.31      1584925.98      6767442.51
      1585148.65      6767756.34
#Sta/Elev= 30
  4644.3 2018.76  4654.1 2019.53  4674.3 2018.19  4694.6 2015.67  4700.5 2014.13
  4705.6 2013.94  4714.8 2012.20  4735.0 2010.28  4763.6 2008.47  4831.8 2006.69
  4876.7 2006.30  4907.1 2004.81  4975.9 2002.88  4976.1 2002.38  4979.6 2002.38
  4979.9 2002.88  5002.7 2003.02  5006.5 2003.43  5012.6 2003.18  5021.2 2003.87
  5042.1 2003.98  5070.7 2006.38  5092.6 2005.28  5113.5 2006.07  5229.2 2007.42
  5300.5 2009.78  5328.2 2011.34  5350.9 2011.37  5371.8 2011.88  5387.5 2012.76
#Mann=3,-1,0
  4644.3    0.05       0  4975.9    0.05       0  4979.9    0.05       0
Bank Sta=4975.9,4979.9
Exp/Cntr=0.3,0.1

Type RM Length L Ch R = 1,176574,76,76,76
BEGIN DESCRIPTION:
Cedar Creek 176574.06
END DESCRIPTION:
XS GIS Cut Line= 4
      1584789.25      6767107.83      1584883.01      6767460.74
      1584918.16      6767523.24      1585104.34      6767782.33
#Sta/Elev= 30
  4635.6 2018.89  4666.8 2017.60  4714.9 2011.71  4755.1 2008.17  4790.1 2006.83
  4870.4 2005.55  4894.4 2006.33  4910.6 2007.89  4915.7 2006.67  4945.5 2007.04
  4950.7 2005.70  4966.9 2006.37  4990.9 2005.72  5014.9 2006.05  5030.8 2007.52
  5036.6 2006.73  5052.5 2008.63  5058.3 2008.29  5066.4 2009.13  5072.3 2006.89
  5080.0 2006.99  5100.9 2003.67  5101.2 2003.17  5104.9 2003.67  5115.6 2005.35
  5159.8 2005.06  5245.8 2006.59  5346.4 2009.01  5382.0 2011.22  5391.5 2010.88
#Mann=3,-1,0
  4635.6    0.05       0  5100.9    0.05       0  5104.9    0.05       0
Bank Sta=5100.9,5104.9
Exp/Cntr=0.3,0.1

Type RM Length L Ch R = 1,176498,187,187,187
BEGIN DESCRIPTION:
Cedar Creek 176497.71
END DESCRIPTION:
XS GIS Cut Line= 4
      1584717.65      6767097.50      1584816.60      6767489.39
      1584875.20      6767580.53      1585083.55      6767852.70
#Sta/Elev= 30
  4599.0 2019.98  4647.7 2015.05  4652.8 2015.19  4671.7 2012.94  4729.8 2008.18
  4811.9 2005.08  4858.1 2004.76  4878.0 2003.56  4888.3 2002.17  4894.0 2000.50
  4929.6 1995.56  4935.0 1994.15  4974.1 1992.41  4974.3 1991.91  4978.1 1992.41
  5014.4 1993.22  5044.8 1998.02  5072.9 2000.82  5087.1 2003.62  5096.3 2004.07
  5158.7 2004.28  5173.2 2005.44  5187.7 2004.60  5302.0 2006.82  5322.8 2007.81
  5337.3 2006.92  5380.9 2008.53  5387.2 2009.49  5416.2 2009.61  5454.3 2011.30
#Mann=3,-1,0
  4599.0    0.05       0  4974.1    0.05       0  4978.1    0.05       0
Bank Sta=4974.1,4978.1
Exp/Cntr=0.3,0.1

Type RM Length L Ch R = 1,176311,76,76,76
BEGIN DESCRIPTION:
Cedar Creek 176311.13
END DESCRIPTION:
XS GIS Cut Line= 5
      1584672.07      6767098.74      1584678.58      6767365.69
      1584700.72      6767514.13      1584785.35      6767561.00
      1585058.78      6767880.00
#Sta/Elev= 30
  4735.9 2019.97  4765.2 2017.92  4815.2 2011.57  4865.2 2006.92  4975.2 2003.58
  5011.4 2003.93  5075.7 1998.68  5086.2 1996.01  5116.5 1995.11  5145.0 1996.06
  5150.0 1994.30  5158.3 1994.95  5165.5 1992.39  5165.7 1991.89  5169.5 1992.39
  5173.2 1993.96  5180.8 1992.79  5189.2 1993.30  5238.4 2001.66  5249.8 2001.89
  5254.6 2003.80  5283.2 2006.73  5297.5 2006.76  5318.3 2002.84  5332.6 2002.35
  5353.4 2003.79  5453.3 2004.39  5552.1 2008.08  5574.0 2007.60  5669.9 2010.35
#Mann=3,-1,0
  4735.9    0.05       0  5165.5    0.05       0  5169.5    0.05       0
Bank Sta=5165.5,5169.5
Exp/Cntr=0.3,0.1

Type RM Length L Ch R = 1,176235,228,228,228
BEGIN DESCRIPTION:
Cedar Creek 176234.52
END DESCRIPTION:
XS GIS Cut Line= 5
      1584582.23      6767093.57      1584610.87      6767343.55
      1584629.10      6767486.78      1584675.98      6767609.18
      1585026.23      6767916.46
#Sta/Elev= 30
  4752.2 2015.75  4786.9 2012.14  4821.3 2010.66  4837.2 2008.82  4978.1 2003.42
  5008.6 2003.99  5048.6 2007.75  5119.2 2010.30  5177.5 2010.14  5182.8 2009.11
  5202.2 2009.59  5207.5 2008.81  5213.8 2009.59  5237.6 2009.35  5291.5 2010.86
  5313.3 2010.09  5320.0 2007.58  5327.5 2008.72  5334.2 2005.19  5341.8 2004.77
  5348.4 2002.50  5370.2 2002.94  5395.8 2002.06  5396.0 2001.56  5399.8 2002.06
  5518.3 2003.69  5597.0 2006.09  5653.0 2006.24  5724.2 2009.67  5745.2 2009.92
#Mann=3,-1,0
  4752.2    0.05       0  5395.8    0.05       0  5399.8    0.05       0
Bank Sta=5395.8,5399.8
Exp/Cntr=0.3,0.1

Type RM Length L Ch R = 1,176007,185,185,185
BEGIN DESCRIPTION:
Cedar Creek 176007.01
END DESCRIPTION:
XS GIS Cut Line= 4
      1584506.71      6767128.70      1584547.07      6767545.38
      1584643.43      6767684.70      1585010.34      6767957.93
#Sta/Elev= 30
  4584.9 2009.82  4704.8 2005.23  4755.0 2003.85  4804.0 2003.19  4823.4 2002.97
  4855.5 2001.60  4925.5 2000.48  5008.7 1997.35  5009.0 1996.85  5012.5 1996.85
  5012.7 1997.35  5046.6 1998.52  5102.0 1998.77  5112.1 1998.84  5118.2 1999.51
  5127.0 1999.13  5168.9 2000.06  5171.9 2000.80  5184.0 2000.98  5190.2 2001.74
  5348.7 2002.57  5411.8 2004.00  5419.6 2003.67  5469.7 2004.43  5475.9 2005.10
  5540.6 2005.99  5569.8 2007.62  5590.6 2007.32  5605.2 2008.75  5630.4 2009.30
#Mann=5,-1,0
  4584.9    0.05       0  4804.0    0.12       0  5008.7    0.07       0
  5012.7    0.12       0  5102.0    0.05       0
Bank Sta=5008.7,5012.7
Exp/Cntr=0.3,0.1

Type RM Length L Ch R = 1,175822,175,175,175
BEGIN DESCRIPTION:
Cedar Creek 175821.96
END DESCRIPTION:
XS GIS Cut Line= 3
      1584392.88      6767171.29      1584396.03      6767539.88
      1584491.73      6768253.80
#Sta/Elev= 30
  4631.4 2008.31  4778.1 2002.80  4818.1 2002.23  4858.1 2000.77  4938.1 1999.76
  4976.1 1996.10  4976.4 1995.60  4979.9 1995.60  4980.1 1996.10  4986.7 1996.33
  5030.7 1996.63  5109.6 1998.44  5119.2 1998.01  5169.6 1998.85  5220.1 2001.54
  5240.2 2000.56  5381.5 2002.81  5462.2 2005.89  5484.5 2005.19  5502.6 2005.50
  5542.9 2007.60  5557.4 2007.93  5563.1 2007.05  5573.2 2007.07  5603.5 2007.86
  5635.4 2009.98  5664.0 2009.19  5694.3 2011.19  5703.3 2010.59  5720.3 2011.13
#Mann=5,-1,0
  4631.4    0.05       0  4976.1    0.07       0  4980.1    0.05       0
  4986.7    0.12       0  5030.7    0.05       0
Bank Sta=4976.1,4980.1
Exp/Cntr=0.3,0.1

Type RM Length L Ch R = 1,175647,219,219,219
BEGIN DESCRIPTION:
Cedar Creek 175647.25
END DESCRIPTION:
XS GIS Cut Line= 3
      1584221.15      6767173.68      1584221.86      6767541.60
      1584268.89      6768623.16
#Sta/Elev= 30
  4633.7 2007.05  4688.0 2003.75  4728.0 2003.25  4758.0 2001.43  4798.0 2001.88
  4848.0 1998.92  4888.0 1999.15  4995.3 1994.16  4995.6 1993.66  4999.3 1994.16
  5133.3 1996.15  5219.4 1998.12  5338.3 2000.35  5448.4 2000.26  5598.6 2004.04
  5618.6 2001.98  5651.5 2005.57  5658.6 2007.97  5688.7 2009.13  5758.7 2007.26
  5778.8 2007.90  5798.8 2002.79  5858.8 2002.93  5881.7 2004.32  5978.9 2005.77
  5989.0 2007.31  6009.0 2007.89  6039.0 2011.77  6059.0 2010.75  6084.2 2014.00
#Mann=5,-1,0
  4633.7    0.05       0  4995.3    0.05       0  4999.3    0.05       0
  5133.3    0.12       0  5219.4    0.05       0
Bank Sta=4995.3,4999.3
Exp/Cntr=0.3,0.1

Type RM Length L Ch R = 1,175428,215,215,215
BEGIN DESCRIPTION:
Cedar Creek 175364.42
END DESCRIPTION:
XS GIS Cut Line= 3
      1584010.65      6767052.14      1584039.84      6767587.35
      1584145.11      6768563.89
#Sta/Elev= 30
  4464.0 2004.53  4530.0 2001.21  4560.0 2001.73  4620.1 1998.88  4660.1 1998.88
  4958.6 1993.00  4958.8 1992.50  4962.6 1993.00  4980.6 1994.11  4997.8 1993.07
  5040.9 1993.29  5131.4 1996.08  5171.6 1996.25  5187.4 1998.15  5201.8 1997.08
  5232.0 1997.70  5272.2 1996.46  5382.9 1997.16  5483.4 1999.87  5543.8 1997.99
  5743.9 1999.47  5775.1 2001.66  5795.2 2000.23  5825.4 2004.82  5840.9 2004.79
  5845.9 2006.15  5932.8 2006.06  5937.8 2007.96  5956.2 2008.30  5982.2 2012.18
#Mann=3,-1,0
  4464.0    0.05       0  4958.6    0.05       0  4962.6    0.05       0
Bank Sta=4958.6,4962.6
Exp/Cntr=0.3,0.1

Type RM Length L Ch R = 1,175213,190,190,190
BEGIN DESCRIPTION:
Cedar Creek 175211.98
END DESCRIPTION:
XS GIS Cut Line= 3
      1583782.78      6767108.56      1583825.68      6767598.08
      1583995.45      6768471.34
#Sta/Elev= 30
  4517.9 1996.68  4577.6 1996.83  4607.7 1995.33  4868.7 1992.21  4918.9 1992.18
  4944.1 1993.40  5004.7 1991.72  5005.0 1991.22  5008.7 1991.72  5085.0 1992.18
  5213.0 1996.52  5263.9 1996.51  5296.8 1998.07  5386.1 2000.12  5498.2 1995.00
  5611.9 1995.92  5630.6 1996.86  5651.0 1999.34  5658.4 1999.09  5663.5 1997.41
  5752.9 1998.21  5761.8 1998.40  5773.3 2000.90  5813.4 2004.89  5818.5 2006.54
  5824.2 2006.49  5834.4 2008.08  5870.2 2009.49  5875.3 2011.14  5898.9 2010.54
#Mann=3,-1,0
  4517.9    0.05       0  5004.7    0.05       0  5008.7    0.05       0
Bank Sta=5004.7,5008.7
Exp/Cntr=0.3,0.1

Type RM Length L Ch R = 1,175023,211,211,211
BEGIN DESCRIPTION:
Cedar Creek 175022.93
END DESCRIPTION:
XS GIS Cut Line= 3
      1583598.33      6767112.92      1583683.66      6767711.74
      1583758.67      6768334.87
#Sta/Elev= 30
  4396.7 1996.56  4412.8 1996.95  4452.3 1994.92  4523.0 1994.56  4620.1 1992.40
  4832.5 1992.31  4886.7 1990.63  4896.8 1991.08  4965.5 1990.16  4965.7 1989.66
  4969.5 1990.16  5028.0 1990.59  5136.0 1994.69  5141.1 1994.25  5189.2 1995.61
  5199.2 1995.11  5305.3 1997.70  5370.5 1994.48  5387.4 1994.62  5392.5 1995.50
  5420.8 1993.98  5469.6 1994.03  5481.3 1995.90  5511.5 1997.21  5541.7 2002.16
  5551.7 2002.92  5556.7 2001.36  5571.9 2004.29  5582.0 2005.28  5629.2 2008.28
#Mann=3,-1,0
  4396.7    0.05       0  4965.5    0.05       0  4969.5    0.05       0
Bank Sta=4965.5,4969.5
Exp/Cntr=0.3,0.1

Type RM Length L Ch R = 1,174812,331,331,331
BEGIN DESCRIPTION:
Cedar Creek 174811.89
END DESCRIPTION:
XS GIS Cut Line= 3
      1583415.16      6767310.66      1583481.53      6767738.04
      1583562.16      6768394.20
#Sta/Elev= 30
  4567.5 1995.37  4655.9 1994.21  4676.1 1992.87  4716.6 1992.25  4807.7 1992.44
  4856.5 1990.98  4979.7 1990.23  4995.5 1989.50  4995.7 1989.00  4999.5 1989.50
  5120.9 1990.38  5171.2 1992.55  5272.0 1994.42  5302.2 1993.40  5311.4 1991.66
  5322.4 1991.47  5332.4 1992.40  5392.7 1992.20  5423.1 1995.63  5453.3 1994.92
  5463.4 1995.97  5523.9 1998.08  5560.3 1997.35  5574.3 1998.40  5584.3 2000.10
  5594.4 2003.01  5604.5 2004.00  5614.6 2001.55  5634.7 1999.29  5661.1 1999.33
#Mann=3,-1,0
  4567.5    0.05       0  4995.5   0.035       0  4999.5    0.05       0
Bank Sta=4995.5,4999.5
Exp/Cntr=0.3,0.1

Type RM Length L Ch R = 1,174481,359,359,359
BEGIN DESCRIPTION:
Cedar Creek 174481
END DESCRIPTION:
XS GIS Cut Line= 3
      1583198.09      6767517.26      1583205.91      6767894.90
      1583217.62      6768208.66
#Sta/Elev= 30
  4624.8 1998.65  4645.5 1998.02  4685.6 1997.79  4718.7 1997.02  4735.6 1995.51
  4745.6 1995.27  4765.6 1992.60  4785.6 1990.92  4815.6 1989.25  4885.6 1987.95
  4945.6 1987.79  4975.6 1988.12  4993.6 1986.83  4993.9 1986.33  4997.4 1986.33
  4997.6 1986.83  5035.6 1987.62  5055.7 1987.20  5105.7 1987.24  5111.4 1987.79
  5116.4 1987.59  5125.7 1988.46  5155.7 1989.29  5175.7 1988.96  5185.7 1989.26
  5205.8 1988.32  5235.8 1988.46  5275.8 1989.46  5285.8 1989.13  5316.5 1989.81
#Mann=3,-1,0
  4624.8    0.05       0  4993.6    0.05       0  4997.6    0.05       0
Bank Sta=4993.6,4997.6
Exp/Cntr=0.3,0.1

Type RM Length L Ch R = 1,174122,364,364,364
BEGIN DESCRIPTION:
Cedar Creek 174121.83
END DESCRIPTION:
XS GIS Cut Line= 3
      1582755.21      6767569.67      1582889.75      6767955.93
      1583160.51      6768597.09
#Sta/Elev= 30
  4592.6 2007.23  4638.0 2005.38  4694.9 1995.00  4700.2 1996.13  4707.3 1994.87
  4726.0 1993.76  4731.3 1996.17  4757.1 1991.89  4770.8 1992.53  4866.1 1987.11
  4982.6 1986.15  4998.1 1985.32  4998.3 1984.82  5002.1 1985.32  5129.7 1986.56
  5153.4 1985.92  5211.7 1987.28  5230.0 1986.10  5275.2 1986.57  5329.5 1987.54
  5341.1 1989.10  5359.4 1988.30  5503.2 1990.72  5517.9 1991.26  5524.9 1992.51
  5541.6 1991.76  5641.9 1994.09  5665.6 1995.59  5687.7 1994.89  5697.6 1995.86
#Mann=3,-1,0
  4592.6    0.05       0  4998.1    0.05       0  5002.1    0.05       0
Bank Sta=4998.1,5002.1
Exp/Cntr=0.3,0.1

Type RM Length L Ch R = 1,173758,327,327,327
BEGIN DESCRIPTION:
Cedar Creek 173758.48
END DESCRIPTION:
XS GIS Cut Line= 3
      1582334.22      6767899.52      1582646.70      6768198.99
      1583140.72      6768790.52
#Sta/Elev= 30
  4568.5 1994.78  4603.3 1994.86  4638.8 1993.33  4709.3 1993.27  4751.8 1991.79
  4872.2 1991.36  4893.3 1989.61  4900.5 1989.94  4907.4 1988.64  4914.7 1990.06
  4921.6 1988.93  4928.8 1990.00  4964.0 1984.50  4995.0 1983.49  4995.2 1982.99
  4999.0 1983.49  5134.0 1985.02  5205.6 1983.98  5255.1 1984.41  5275.9 1986.05
  5361.8 1987.47  5382.6 1989.40  5390.4 1988.46  5468.5 1990.13  5482.1 1990.67
  5495.9 1992.60  5645.5 1993.52  5674.1 1995.36  5688.5 1994.40  5772.0 1996.95
#Mann=3,-1,0
  4568.5    0.05       0  4995.0   0.035       0  4999.0    0.05       0
Bank Sta=4995,4999
Exp/Cntr=0.3,0.1

Type RM Length L Ch R = 1,173431,328,328,328
BEGIN DESCRIPTION:
Cedar Creek 173431.06
END DESCRIPTION:
XS GIS Cut Line= 3
      1582161.92      6768259.23      1582444.44      6768446.71
      1582888.46      6768701.92
#Sta/Elev= 30
  4660.1 1984.99  4698.4 1985.77  4725.5 1985.36  4755.6 1985.76  4761.6 1985.29
  4791.7 1985.72  4842.8 1985.52  4927.8 1983.35  4996.5 1982.25  5008.7 1982.21
  5022.9 1982.88  5030.3 1982.25  5036.0 1982.58  5043.9 1982.12  5044.2 1981.62
  5047.7 1981.62  5047.9 1982.12  5051.8 1983.11  5073.4 1982.88  5080.5 1983.37
  5234.4 1983.19  5277.5 1984.75  5299.7 1984.80  5330.7 1986.48  5395.4 1986.53
  5411.2 1987.39  5426.6 1989.56  5432.8 1988.07  5448.6 1987.70  5511.3 1988.73
#Mann=3,-1,0
  4660.1    0.05       0  5043.9   0.035       0  5047.9    0.05       0
Bank Sta=5043.9,5047.9
Exp/Cntr=0.3,0.1

Type RM Length L Ch R = 1,173103,594,594,594
BEGIN DESCRIPTION:
Cedar Creek 173102.51
END DESCRIPTION:
XS GIS Cut Line= 3
      1582101.16      6768617.40      1582311.63      6768731.86
      1582841.44      6768999.37
#Sta/Elev= 30
  4758.4 1982.67  4851.0 1981.40  4980.1 1980.85  4980.3 1980.35  4983.8 1980.35
  4984.1 1980.85  5013.0 1981.93  5042.9 1981.72  5048.5 1982.14  5057.8 1981.49
  5087.5 1981.67  5109.8 1981.12  5154.4 1981.48  5199.0 1982.96  5271.5 1984.12
  5304.2 1985.21  5310.5 1986.09  5338.4 1985.97  5383.0 1987.41  5393.8 1988.13
  5405.3 1990.82  5422.0 1988.77  5472.3 1990.28  5511.1 1990.62  5527.8 1991.66
  5533.4 1991.44  5539.5 1992.48  5555.7 1993.26  5572.4 1992.02  5591.5 1992.43
#Mann=3,-1,0
  4758.4    0.05       0  4980.1   0.035       0  4984.1    0.05       0
Bank Sta=4980.1,4984.1
Exp/Cntr=0.3,0.1

Type RM Length L Ch R = 1,172509,555,555,555
BEGIN DESCRIPTION:
Cedar Creek 172509.19
END DESCRIPTION:
XS GIS Cut Line= 3
      1581717.42      6769256.38      1582130.80      6769264.31
      1582951.87      6769292.03
#Sta/Elev= 30
  4588.0 1979.95  4685.6 1980.55  4765.6 1979.69  4795.6 1980.09  4865.6 1978.29
  4895.6 1978.82  4905.6 1977.80  4936.8 1977.91  4955.6 1976.99  4985.7 1977.94
  5006.1 1977.61  5013.7 1976.42  5013.9 1975.92  5017.7 1976.42  5025.7 1977.41
  5065.7 1978.39  5259.9 1980.09  5275.8 1980.97  5295.8 1980.51  5315.8 1981.65
  5395.9 1983.04  5435.9 1984.80  5455.9 1986.61  5465.9 1986.27  5526.0 1988.85
  5536.0 1988.39  5566.0 1989.71  5586.0 1989.13  5686.0 1993.44  5823.0 1997.67
#Mann=3,-1,0
  4588.0    0.05       0  5013.7   0.035       0  5017.7    0.05       0
Bank Sta=5013.7,5017.7
Exp/Cntr=0.3,0.1

Type RM Length L Ch R = 1,171954,532,532,532
BEGIN DESCRIPTION:
Cedar Creek 171954.37
END DESCRIPTION:
XS GIS Cut Line= 4
      1581431.00      6769313.02      1581475.23      6769480.22
      1581750.36      6769642.90      1582571.64      6769968.64
#Sta/Elev= 30
  4508.0 1976.41  4575.2 1975.58  4647.6 1973.11  4668.3 1973.55  4686.5 1971.96
  4702.1 1972.83  4707.9 1971.91  4723.5 1972.50  4750.8 1971.74  4926.3 1972.18
  4969.1 1970.83  4969.4 1970.33  4973.1 1970.83  5016.3 1972.16  5263.8 1974.36
  5324.6 1975.80  5339.1 1977.46  5392.9 1976.80  5425.1 1977.84  5438.0 1979.29
  5457.0 1978.37  5511.0 1981.42  5565.0 1981.47  5586.5 1983.87  5608.0 1983.24
  5672.6 1986.22  5694.1 1985.95  5780.1 1989.76  5801.7 1989.18  5884.1 1992.42
#Mann=3,-1,0
  4508.0    0.05       0  4969.1   0.035       0  4973.1    0.05       0
Bank Sta=4969.1,4973.1
Exp/Cntr=0.3,0.1

Type RM Length L Ch R = 1,171422,445,445,445
BEGIN DESCRIPTION:
Cedar Creek 171422.63
END DESCRIPTION:
XS GIS Cut Line= 3
      1580480.44      6769202.32      1581265.35      6769790.18
      1581758.84      6770072.74
#Sta/Elev= 30
  4020.3 1972.09  4049.8 1971.17  4156.0 1971.12  4320.7 1968.96  4335.2 1969.75
  4370.7 1967.64  4426.9 1966.98  4463.3 1965.29  4520.7 1965.55  4539.5 1964.40
  4539.8 1963.90  4543.5 1964.40  4570.7 1965.63  4691.6 1965.47  4763.1 1966.51
  4835.3 1966.31  4963.0 1967.51  4970.8 1966.49  5006.5 1967.38  5108.6 1967.76
  5277.1 1969.79  5300.1 1969.27  5344.6 1970.41  5357.8 1969.81  5452.5 1971.08
  5474.1 1972.33  5496.0 1971.88  5519.1 1973.43  5542.1 1972.79  5569.6 1974.00
#Mann=3,-1,0
  4020.3    0.05       0  4539.5   0.035       0  4543.5    0.05       0
Bank Sta=4539.5,4543.5
Exp/Cntr=0.3,0.1

Type RM Length L Ch R = 1,170977,403,403,403
BEGIN DESCRIPTION:
Cedar Creek 170977.49
END DESCRIPTION:
XS GIS Cut Line= 3
      1580435.66      6769576.45      1580883.62      6769809.54
      1581617.98      6770171.51
#Sta/Elev= 30
  4495.5 1970.96  4539.8 1970.40  4554.9 1970.98  4615.6 1968.97  4681.9 1969.07
  4704.0 1967.73  4754.0 1967.43  4770.3 1966.64  4776.6 1964.48  4786.8 1964.16
  4956.9 1964.11  4985.7 1964.97  5004.0 1964.69  5011.5 1963.39  5011.8 1962.89
  5015.5 1963.39  5068.9 1965.17  5135.8 1964.98  5470.3 1967.11  5492.6 1968.45
  5502.0 1967.56  5552.5 1968.28  5581.8 1969.75  5597.4 1969.17  5614.3 1970.51
  5626.3 1969.77  5726.6 1970.55  5754.6 1971.96  5805.1 1971.82  5819.2 1972.49
#Mann=3,-1,0
  4495.5    0.05       0  5011.5   0.035       0  5015.5    0.05       0
Bank Sta=5011.5,5015.5
Exp/Cntr=0.3,0.1

Type RM Length L Ch R = 1,170574,465,465,465
BEGIN DESCRIPTION:
Cedar Creek 170573.61
END DESCRIPTION:
XS GIS Cut Line= 3
      1580186.15      6769820.40      1580639.26      6770102.94
      1581509.69      6770393.09
#Sta/Elev= 30
  4466.1 1971.42  4559.0 1970.63  4607.7 1968.78  4769.3 1966.57  4848.4 1964.39
  4854.3 1962.86  4863.7 1962.94  4869.6 1961.52  4885.0 1961.80  4888.8 1960.83
  4889.1 1960.33  4893.0 1960.83  4906.2 1960.83  4921.5 1962.76  5016.7 1961.92
  5037.8 1960.88  5158.7 1962.91  5185.0 1962.27  5285.2 1963.46  5354.0 1963.10
  5522.6 1965.76  5538.2 1966.85  5543.7 1965.97  5569.8 1966.25  5607.0 1968.10
  5670.2 1968.05  5733.5 1970.07  5775.6 1969.51  5838.9 1971.52  5917.6 1972.46
#Mann=3,-1,0
  4466.1    0.05       0  4888.8   0.035       0  4893.0    0.05       0
Bank Sta=4888.8,4893
Exp/Cntr=0.3,0.1

Type RM Length L Ch R = 1,170109,408,408,408
BEGIN DESCRIPTION:
Cedar Creek 170109.09
END DESCRIPTION:
XS GIS Cut Line= 3
      1579952.73      6770356.42      1580650.63      6770392.87
      1581626.37      6770509.20
#Sta/Elev= 30
  4299.1 1969.03  4431.5 1968.87  4621.9 1964.58  4681.9 1964.29  4701.9 1962.98
  4742.0 1963.03  4762.0 1961.55  4952.3 1959.96  5001.1 1958.16  5001.4 1957.66
  5005.3 1958.16  5022.5 1960.18  5032.6 1959.60  5324.6 1963.33  5354.8 1964.65
  5455.5 1965.48  5475.7 1966.61  5516.0 1966.35  5556.2 1968.08  5576.4 1967.33
  5636.8 1968.38  5667.0 1970.15  5707.3 1969.79  5756.0 1971.78  5828.2 1972.25
  5843.5 1973.65  5858.4 1973.01  5918.8 1974.13  5949.0 1976.55  5980.6 1976.17
#Mann=3,-1,0
  4299.1    0.05       0  5001.1   0.035       0  5005.3    0.05       0
Bank Sta=5001.1,5005.3
Exp/Cntr=0.3,0.1

Type RM Length L Ch R = 1,169701,641,641,641
BEGIN DESCRIPTION:
Cedar Creek 169701.02
END DESCRIPTION:
XS GIS Cut Line= 3
      1579886.54      6770562.66      1580702.54      6770784.89
      1581339.67      6770984.53
#Sta/Elev= 30
  4155.0 1969.15  4288.1 1968.19  4311.3 1968.79  4345.9 1967.10  4425.4 1966.34
  4465.1 1963.99  4485.1 1964.24  4516.2 1962.58  4579.2 1962.64  4827.1 1957.24
  4899.6 1958.49  4930.7 1957.17  4961.8 1958.78  5028.7 1958.34  5043.1 1956.34
  5043.4 1955.84  5047.3 1956.34  5076.7 1958.85  5087.1 1958.65  5131.2 1961.54
  5190.9 1961.98  5254.8 1965.17  5293.4 1964.83  5325.9 1966.57  5363.6 1966.43
  5380.6 1968.24  5412.0 1967.94  5443.4 1970.16  5525.8 1970.30  5668.4 1973.91
#Mann=3,-1,0
  4155.0    0.05       0  5043.1   0.035       0  5047.3    0.05       0
Bank Sta=5043.1,5047.3
Exp/Cntr=0.3,0.1

Type RM Length L Ch R = 1,169060,497,497,497
BEGIN DESCRIPTION:
Cedar Creek 169059.99
END DESCRIPTION:
XS GIS Cut Line= 3
      1579796.49      6770862.93      1580447.55      6771188.46
      1580998.06      6771393.60
#Sta/Elev= 30
  4270.2 1967.67  4311.4 1967.44  4361.7 1964.12  4428.8 1961.99  4490.3 1961.23
  4652.4 1956.75  4794.0 1955.81  4870.4 1956.62  4943.1 1955.69  4965.4 1953.97
  5005.9 1954.54  5014.5 1953.60  5014.8 1953.10  5018.9 1953.60  5036.2 1953.83
  5066.6 1959.08  5096.9 1960.79  5187.9 1961.46  5243.2 1963.36  5304.9 1964.06
  5323.5 1965.26  5328.8 1964.67  5400.9 1966.77  5414.5 1967.92  5432.9 1967.17
  5454.3 1969.03  5469.8 1968.02  5530.5 1969.14  5550.1 1970.44  5585.6 1970.46
#Mann=3,-1,0
  4270.2    0.05       0  5014.5   0.035       0  5018.9    0.05       0
Bank Sta=5014.5,5018.9
Exp/Cntr=0.3,0.1

Type RM Length L Ch R = 1,168563,535,535,535
BEGIN DESCRIPTION:
Cedar Creek 168563.41
END DESCRIPTION:
XS GIS Cut Line= 3
      1579705.34      6771063.44      1580179.32      6771511.38
      1580771.55      6771817.88
#Sta/Elev= 30
  4346.9 1967.49  4378.1 1967.47  4406.4 1964.16  4434.7 1962.77  4604.6 1958.47
  4611.5 1959.36  4618.8 1959.16  4625.7 1960.75  4633.0 1960.87  4639.8 1961.99
  4717.9 1963.68  4753.1 1961.52  4767.3 1958.34  4781.4 1956.62  4809.8 1954.79
  4845.0 1953.91  4951.3 1953.37  4977.1 1951.09  4977.4 1950.59  4981.2 1950.59
  4981.5 1951.09  4986.5 1952.65  5029.0 1953.10  5084.1 1955.11  5134.0 1955.13
  5239.1 1959.99  5416.2 1963.08  5432.7 1963.98  5571.2 1965.33  5665.9 1967.38
#Mann=3,-1,0
  4346.9    0.05       0  4977.1   0.035       0  4981.5    0.05       0
Bank Sta=4977.1,4981.5
Exp/Cntr=0.3,0.1

Type RM Length L Ch R = 1,168028,187,187,187
BEGIN DESCRIPTION:
Cedar Creek 168329.457
END DESCRIPTION:
XS GIS Cut Line= 3
      1579786.11      6771362.97      1580107.35      6771943.97
      1580780.45      6772034.76
#Sta/Elev= 30
  4336.1 1966.16  4383.7 1965.99  4448.9 1963.29  4524.6 1958.18  4568.1 1954.07
  4611.6 1952.77  4774.3 1950.50  4913.2 1951.30  4920.9 1950.98  4926.6 1949.30
  4940.4 1948.65  4940.7 1948.15  4944.8 1948.65  4948.3 1950.00  4958.7 1949.29
  4980.4 1950.81  4986.1 1952.38  4999.4 1952.06  5007.7 1954.94  5017.8 1956.20
  5048.1 1957.35  5270.1 1960.66  5280.2 1960.15  5293.6 1957.55  5300.3 1957.52
  5340.7 1961.44  5366.4 1962.15  5371.4 1961.41  5439.1 1963.79  5679.2 1967.83
#Mann=3,-1,0
  4336.1    0.05       0  4940.4   0.035       0  4944.8    0.05       0
Bank Sta=4940.4,4944.8
Exp/Cntr=0.3,0.1

Type RM Length L Ch R = 1,167841,386,386,386
BEGIN DESCRIPTION:
Cedar Creek 167840.838
END DESCRIPTION:
XS GIS Cut Line= 3
      1579648.07      6771383.77      1579979.65      6772037.37
      1580293.55      6772674.32
#Sta/Elev= 30
  4267.1 1965.95  4327.9 1964.82  4341.2 1965.41  4395.2 1962.94  4408.0 1963.68
  4440.0 1960.93  4462.5 1960.82  4474.8 1958.51  4497.1 1957.81  4513.7 1955.69
  4580.5 1952.39  4899.8 1949.76  4936.7 1950.62  4975.7 1949.61  4981.3 1950.38
  4989.5 1948.64  5001.0 1948.48  5001.4 1947.98  5006.0 1948.48  5020.4 1950.81
  5034.1 1951.18  5078.7 1951.43  5093.4 1952.48  5115.8 1950.21  5138.3 1950.61
  5145.6 1952.59  5301.7 1956.12  5407.8 1955.96  5570.6 1957.99  5710.1 1956.75
#Mann=3,-1,0
  4267.1    0.05       0  5001.0   0.035       0  5006.0    0.05       0
Bank Sta=5001,5006
Exp/Cntr=0.3,0.1

Type RM Length L Ch R = 1,167455,1312,1312,1312
BEGIN DESCRIPTION:
Cedar Creek 167454.52
END DESCRIPTION:
XS GIS Cut Line= 3
      1579311.95      6771783.74      1579693.90      6772249.01
      1580155.72      6772877.51
#Sta/Elev= 30
  4396.9 1957.71  4430.1 1957.83  4508.3 1955.49  4586.5 1954.78  4600.8 1953.61
  4664.7 1953.04  4686.9 1951.77  4829.0 1950.54  4907.0 1947.45  4984.6 1949.07
  4991.9 1948.57  4993.3 1946.44  4993.6 1945.94  4998.3 1946.44  5006.5 1947.50
  5012.7 1949.46  5034.8 1948.68  5207.1 1948.48  5248.8 1949.50  5278.1 1949.23
  5284.3 1950.09  5307.4 1949.71  5349.1 1951.04  5357.5 1952.00  5399.3 1952.50
  5413.9 1951.99  5434.8 1952.95  5585.2 1953.54  5664.7 1951.97  5778.8 1953.51
#Mann=3,-1,0
  4396.9    0.05       0  4993.3   0.035       0  4998.3    0.05       0
Bank Sta=4993.3,4998.3
Exp/Cntr=0.3,0.1

Type RM Length L Ch R = 1,166143,390,390,390
BEGIN DESCRIPTION:
Cedar Creek 166143.3
END DESCRIPTION:
XS GIS Cut Line= 3
      1579319.24      6772348.05      1579301.88      6773198.72
      1579353.92      6774764.31
#Sta/Elev= 30
  4157.2 1949.68  4467.2 1946.98  4647.3 1946.79  4717.3 1945.88  4757.3 1943.63
  4777.3 1945.40  4877.3 1945.32  4917.3 1943.64  4927.3 1944.05  4997.3 1942.28
  5005.2 1940.69  5010.2 1940.69  5014.5 1938.01  5014.9 1937.51  5020.2 1938.01
  5027.3 1940.67  5047.3 1943.93  5137.4 1942.09  5197.4 1942.39  5247.4 1941.60
  5277.5 1943.07  5317.5 1947.41  5337.5 1948.05  5553.0 1948.32  5657.7 1950.17
  5907.8 1949.27  6154.2 1950.70  6228.0 1952.25  6454.8 1951.20  6574.5 1951.74
#Mann=3,-1,0
  4157.2    0.05       0  5014.5    0.05       0  5020.2    0.05       0
Bank Sta=5014.5,5020.2
Exp/Cntr=0.3,0.1

Type RM Length L Ch R = 1,165753,526,526,526
BEGIN DESCRIPTION:
Cedar Creek 165753.24
END DESCRIPTION:
XS GIS Cut Line= 3
      1578919.94      6772426.13      1578950.32      6773294.21
      1578937.30      6774782.94
#Sta/Elev= 30
  4136.6 1945.36  4608.8 1944.28  4748.8 1941.33  4788.9 1941.46  4838.9 1939.73
  4888.9 1940.29  4908.9 1942.09  4929.0 1941.59  4939.0 1944.47  4949.0 1943.76
  4969.0 1938.47  4979.0 1936.96  4989.0 1937.49  4991.5 1936.79  4992.0 1936.29
  4998.6 1936.79  5009.6 1937.98  5037.8 1944.30  5049.0 1941.66  5119.0 1940.11
  5339.0 1942.53  5369.0 1943.81  5449.0 1942.03  5509.0 1943.42  5889.0 1944.91
  5939.0 1944.40  6049.0 1946.37  6189.6 1946.53  6249.0 1947.75  6494.0 1947.95
#Mann=3,-1,0
  4136.6    0.05       0  4991.5   0.035       0  4998.6    0.05       0
Bank Sta=4991.5,4998.6
Exp/Cntr=0.3,0.1

Type RM Length L Ch R = 1,165227,725,725,725
BEGIN DESCRIPTION:
Cedar Creek 165226.6
END DESCRIPTION:
XS GIS Cut Line= 3
      1578412.13      6772769.09      1578455.53      6773394.04
      1578568.27      6774634.17
#Sta/Elev= 30
  4374.3 1939.90  4563.7 1941.85  4583.7 1940.67  4603.8 1941.67  4714.0 1938.78
  4784.2 1938.31  4814.3 1939.52  4904.5 1938.42  4964.6 1939.44  4974.7 1938.67
  4984.7 1935.54  4996.7 1933.54  4997.2 1933.04  5003.8 1933.54  5024.8 1934.85
  5044.9 1942.05  5050.0 1945.74  5065.0 1945.70  5075.0 1940.95  5105.1 1937.52
  5125.2 1939.93  5145.3 1938.55  5195.5 1937.94  5406.4 1939.80  5717.8 1939.42
  5777.9 1938.36  5938.7 1939.58  6008.9 1942.76  6109.3 1942.20  6246.0 1943.56
#Mann=3,-1,0
  4374.3    0.05       0  4996.7    0.05       0  5003.8    0.05       0
Bank Sta=4996.7,5003.8
Exp/Cntr=0.3,0.1

Type RM Length L Ch R = 1,164502,413,413,413
BEGIN DESCRIPTION:
Cedar Creek 164501.71
END DESCRIPTION:
XS GIS Cut Line= 6
      1577719.19      6772997.49      1577635.86      6773265.71
      1577695.32      6773495.21      1577805.93      6773641.72
      1577974.32      6773825.68      1578346.66      6774333.24
#Sta/Elev= 30
  4297.6 1937.62  4859.7 1936.21  4918.0 1935.17  4974.2 1936.24  4988.7 1932.76
  5006.2 1931.91  5006.7 1931.41  5013.3 1931.91  5024.0 1932.07  5045.6 1939.50
  5059.7 1939.58  5073.9 1936.34  5088.1 1935.27  5094.9 1936.35  5102.3 1934.98
  5109.1 1934.98  5116.1 1932.18  5123.2 1936.49  5130.0 1936.72  5172.6 1937.15
  5194.2 1934.75  5208.3 1935.85  5253.1 1934.91  5337.3 1936.27  5408.3 1935.27
  5443.9 1936.62  5514.9 1937.10  5558.8 1936.08  5665.4 1936.25  5878.0 1939.90
#Mann=3,-1,0
  4297.6    0.05       0  5006.2    0.05       0  5013.3    0.05       0
Bank Sta=5006.2,5013.3
Exp/Cntr=0.3,0.1

Type RM Length L Ch R = 1,164089,383,383,383
BEGIN DESCRIPTION:
Cedar Creek 164088.9
END DESCRIPTION:
XS GIS Cut Line= 6
      1577487.41      6773031.35      1577323.36      6773229.25
      1577289.50      6773445.40      1577458.71      6773641.72
      1577636.35      6773917.36      1578008.28      6774323.03
#Sta/Elev= 30
  4265.6 1936.08  4463.9 1934.52  4632.7 1933.96  4896.0 1934.58  4931.1 1935.13
  4953.1 1934.75  4973.9 1933.23  4978.0 1932.06  4978.5 1931.56  4984.6 1931.56
  4985.1 1932.06  4988.2 1933.64  5000.6 1934.21  5090.4 1933.64  5198.4 1934.30
  5220.4 1933.74  5226.3 1934.45  5241.5 1934.34  5247.5 1934.86  5277.8 1933.96
  5305.5 1934.43  5349.2 1933.44  5448.5 1933.22  5512.0 1933.92  5540.4 1933.70
  5554.6 1934.31  5618.1 1934.15  5639.7 1934.76  5780.9 1935.21  5878.9 1936.36
#Mann=3,-1,0
  4265.6    0.05       0  4978.0   0.035       0  4985.1    0.05       0
Bank Sta=4978,4985.1
Exp/Cntr=0.3,0.1

Type RM Length L Ch R = 1,163706,365,365,365
BEGIN DESCRIPTION:
Cedar Creek 163705.83
END DESCRIPTION:
XS GIS Cut Line= 5
      1577177.53      6773250.07      1577084.88      6773730.68
      1577316.35      6773973.32      1577618.49      6774262.32
      1577867.67      6774325.62
#Sta/Elev= 30
  4174.2 1933.32  4371.6 1933.49  4641.1 1932.37  4746.6 1932.78  4888.2 1931.42
  4959.0 1932.33  4965.9 1931.65  4969.6 1930.07  4970.1 1929.57  4976.2 1929.57
  4976.7 1930.07  4980.0 1931.58  4987.3 1932.79  5065.1 1931.99  5149.7 1932.47
  5171.1 1931.94  5185.3 1930.72  5199.4 1932.11  5220.5 1932.46  5241.9 1931.80
  5263.0 1932.52  5376.2 1932.44  5516.7 1933.98  5542.1 1934.79  5557.9 1934.35
  5568.3 1935.39  5583.0 1934.15  5599.2 1935.03  5609.5 1934.63  5674.2 1935.50
#Mann=3,-1,0
  4174.2    0.05       0  4969.6   0.035       0  4976.7    0.05       0
Bank Sta=4969.6,4976.7
Exp/Cntr=0.3,0.1

Type RM Length L Ch R = 1,163341,429,429,429
BEGIN DESCRIPTION:
Cedar Creek 163341.12
END DESCRIPTION:
XS GIS Cut Line= 6
      1577062.95      6773388.97      1576911.90      6773665.02
      1576893.67      6773816.06      1577083.71      6774211.17
      1577488.12      6774353.12      1577768.67      6774412.41
#Sta/Elev= 30
  4093.4 1932.59  4305.5 1932.25  4377.3 1931.18  4652.0 1930.30  4702.6 1930.97
  4992.2 1931.60  5006.3 1931.29  5012.7 1929.92  5019.7 1927.16  5020.2 1926.66
  5026.4 1926.66  5026.9 1927.16  5032.5 1929.81  5037.8 1931.17  5076.3 1929.98
  5156.5 1931.06  5161.8 1929.85  5187.5 1931.50  5218.5 1931.09  5275.2 1931.92
  5330.7 1931.72  5351.9 1931.02  5368.2 1932.01  5399.2 1931.16  5446.6 1932.04
  5479.8 1931.60  5548.8 1932.05  5661.2 1933.45  5691.9 1934.15  5716.1 1935.83
#Mann=3,-1,0
  4093.4    0.05       0  5019.7    0.05       0  5026.9    0.05       0
Bank Sta=5019.7,5026.9
Exp/Cntr=0.3,0.1

Type RM Length L Ch R = 1,162912,225,225,225
BEGIN DESCRIPTION:
Cedar Creek 162911.5
END DESCRIPTION:
XS GIS Cut Line= 6
      1576831.17      6773696.26      1576667.93      6774167.16
      1576855.56      6774499.25      1576977.08      6774533.97
      1577346.88      6774518.56      1577770.65      6774508.78
#Sta/Elev= 30
  4120.3 1930.64  4333.1 1929.76  4386.7 1928.61  4616.5 1928.37  4814.9 1929.53
  4904.3 1929.02  4931.7 1930.61  4963.5 1928.32  4969.2 1929.30  5002.4 1928.53
  5010.8 1926.86  5011.3 1926.36  5018.1 1926.86  5041.1 1928.83  5103.5 1928.11
  5121.1 1928.86  5124.7 1927.63  5149.6 1928.54  5154.6 1927.94  5174.5 1929.12
  5264.5 1929.53  5334.6 1929.52  5364.6 1928.00  5394.8 1930.15  5454.7 1930.31
  5484.7 1929.10  5884.8 1933.57  5894.8 1933.96  5914.9 1936.40  5920.5 1936.02
#Mann=3,-1,0
  4120.3    0.05       0  5010.8   0.035       0  5018.1    0.05       0
Bank Sta=5010.8,5018.1
Exp/Cntr=0.3,0.1

Type RM Length L Ch R = 1,162687,172,172,172
BEGIN DESCRIPTION:
Cedar Creek 162687.04
END DESCRIPTION:
XS GIS Cut Line= 6
      1576708.78      6773865.52      1576600.78      6774173.46
      1576827.78      6774714.52      1576951.04      6774719.73
      1576982.29      6774639.87      1577768.68      6774610.33
#Sta/Elev= 30
  4077.1 1929.15  4185.7 1928.21  4485.6 1927.96  4678.1 1929.09  4779.9 1928.35
  4873.1 1930.81  4917.2 1930.88  4939.6 1929.04  4956.3 1929.88  4961.9 1928.80
  4969.8 1929.98  4988.3 1927.87  4988.8 1927.37  4995.9 1927.87  5016.4 1931.84
  5039.4 1931.84  5051.3 1933.62  5072.8 1934.06  5082.7 1934.01  5088.0 1932.86
  5114.7 1933.37  5131.0 1935.52  5221.2 1934.10  5230.0 1930.74  5240.1 1928.49
  5305.0 1929.49  5562.8 1929.30  5751.3 1932.72  5891.3 1933.02  6005.0 1936.78
#Mann=3,-1,0
  4077.1    0.05       0  4988.3   0.035       0  4995.9    0.05       0
Bank Sta=4988.3,4995.9
Exp/Cntr=0.3,0.1

Type RM Length L Ch R = 1,162515,250,250,250
BEGIN DESCRIPTION:
Cedar Creek 162514.96
END DESCRIPTION:
XS GIS Cut Line= 6
      1576648.89      6773909.78      1576561.16      6774265.34
      1576803.47      6774811.75      1576966.67      6774836.05
      1577048.26      6774711.05      1577766.07      6774691.06
#Sta/Elev= 30
  4227.4 1928.69  4623.5 1927.42  4784.6 1927.93  4827.2 1926.94  4950.3 1927.70
  4997.3 1927.29  5026.2 1924.74  5041.5 1926.70  5047.4 1925.21  5055.7 1926.63
  5062.7 1926.53  5095.4 1924.39  5095.9 1923.89  5103.0 1924.39  5105.1 1925.38
  5126.6 1925.39  5135.7 1927.03  5141.6 1925.81  5162.8 1927.69  5223.6 1927.46
  5233.7 1928.21  5294.4 1928.88  5343.0 1928.49  5399.8 1929.30  5475.5 1929.29
  5482.5 1928.25  5781.6 1929.66  5982.0 1933.57  6162.2 1935.19  6243.3 1937.53
#Mann=3,-1,0
  4227.4    0.05       0  5095.4   0.035       0  5103.0    0.05       0
Bank Sta=5095.4,5103
Exp/Cntr=0.3,0.1

Type RM Length L Ch R = 1,162265,321,321,321
BEGIN DESCRIPTION:
Mapping XS 271cfcc5
END DESCRIPTION:
XS GIS Cut Line= 4
      1576607.69      6773912.83      1576459.24      6774379.01
      1576467.05      6775248.80      1576604.63      6775523.95
#Sta/Elev= 30
  4293.7 1928.39  4413.6 1927.73  4445.8 1928.06  4585.2 1927.49  4760.9 1927.23
  4811.9 1927.75  4921.9 1927.33  4961.9 1925.97  4971.9 1925.20  4988.1 1923.06
  4988.6 1922.56  4995.2 1922.56  4995.7 1923.06  5001.9 1925.04  5011.9 1926.51
  5021.9 1926.75  5041.9 1925.93  5091.9 1925.67  5171.9 1926.59  5222.0 1925.50
  5272.0 1927.36  5322.0 1928.10  5342.0 1927.60  5382.0 1928.71  5492.0 1928.77
  5622.0 1930.22  5686.4 1929.95  5830.8 1930.80  5897.8 1930.53  5960.4 1931.33
#Mann=3,-1,0
  4293.7    0.05       0  4988.1   0.035       0  4995.7    0.05       0
Bank Sta=4988.1,4995.7
Exp/Cntr=0.3,0.1

Type RM Length L Ch R = 1,161944,318,318,318
BEGIN DESCRIPTION:
Mapping XS 6bf77e58
END DESCRIPTION:
XS GIS Cut Line= 4
      1576537.38      6773897.22      1576253.51      6774334.74
      1576118.10      6775037.86      1576302.65      6775453.76
#Sta/Elev= 30
  4263.0 1928.05  4403.1 1927.47  4424.2 1927.86  4460.5 1927.09  4475.6 1927.34
  4502.7 1926.49  4620.6 1926.09  4626.6 1925.66  4662.8 1925.49  4777.5 1925.46
  4855.0 1926.02  4920.3 1924.74  4963.9 1925.44  5001.7 1925.06  5010.7 1925.52
  5012.0 1922.98  5012.5 1922.48  5019.1 1922.48  5019.6 1922.98  5022.1 1923.96
  5032.3 1925.38  5042.5 1925.50  5154.5 1925.40  5185.0 1924.97  5223.4 1925.42
  5256.3 1924.33  5286.9 1924.17  5368.3 1925.48  5778.1 1927.89  5955.6 1928.33
#Mann=3,-1,0
  4263.0    0.05       0  5012.0    0.05       0  5019.6    0.05       0
Bank Sta=5012,5019.6
Exp/Cntr=0.3,0.1

Type RM Length L Ch R = 1,161626,580,580,580
BEGIN DESCRIPTION:
Mapping XS 02f155db
END DESCRIPTION:
XS GIS Cut Line= 4
      1576391.53      6773915.47      1575961.85      6774261.82
      1575836.85      6774889.42      1576050.19      6775409.76
#Sta/Elev= 30
  4219.2 1926.54  4438.9 1924.59  4781.5 1923.24  4827.5 1923.61  4934.8 1923.58
  4960.9 1923.99  4971.1 1924.56  4980.8 1924.34  4985.9 1923.72  4991.5 1922.44
  5001.7 1922.00  5011.9 1924.44  5052.7 1924.25  5062.9 1924.77  5088.1 1923.86
  5134.0 1923.66  5175.1 1924.45  5215.8 1924.70  5277.0 1923.44  5314.0 1921.87
  5314.5 1921.37  5321.1 1921.37  5321.6 1921.87  5358.6 1922.25  5394.6 1923.63
  5399.7 1923.44  5417.1 1924.07  5470.5 1924.92  5831.0 1925.13  5973.4 1926.12
#Mann=3,-1,0
  4219.2    0.05       0  5314.0    0.05       0  5321.6    0.05       0
Bank Sta=5314,5321.6
Exp/Cntr=0.3,0.1

Type RM Length L Ch R = 1,161046,303,303,303
BEGIN DESCRIPTION:
Mapping XS 2d25a07f
END DESCRIPTION:
XS GIS Cut Line= 4
      1575188.44      6774089.96      1575352.47      6774188.90
      1575438.41      6774566.51      1575805.32      6775123.37
#Sta/Elev= 30
  4655.8 1934.62  4659.7 1933.72  4665.5 1933.19  4681.0 1934.67  4686.9 1934.35
  4696.5 1933.30  4710.2 1930.09  4717.9 1928.79  4723.7 1927.02  4776.1 1923.57
  4827.0 1922.44  4881.8 1922.00  4887.5 1922.58  4938.7 1921.17  4949.0 1921.28
  4967.9 1922.53  4994.5 1920.09  4995.0 1919.59  5005.5 1919.59  5006.0 1920.09
  5010.5 1922.27  5021.2 1922.81  5255.0 1920.70  5276.1 1921.07  5284.3 1921.66
  5348.4 1921.03  5441.7 1922.40  5535.8 1922.64  5580.3 1923.55  5901.5 1924.64
#Mann=3,-1,0
  4655.8    0.05       0  4994.5    0.05       0  5006.0    0.05       0
Bank Sta=4994.5,5006
Exp/Cntr=0.3,0.1

Type RM Length L Ch R = 1,160743,425,425,425
BEGIN DESCRIPTION:
Cedar Creek 160743.08
END DESCRIPTION:
XS GIS Cut Line= 3
      1574841.58      6774132.00      1575100.25      6774395.88
      1575742.60      6775161.49
#Sta/Elev= 30
  4630.8 1934.70  4637.5 1933.49  4644.5 1934.38  4651.7 1933.47  4658.7 1933.94
  4665.8 1932.35  4672.8 1932.91  4679.9 1931.21  4686.9 1932.27  4694.1 1931.33
  4701.1 1931.79  4715.2 1930.23  4722.4 1928.42  4729.4 1928.82  4743.5 1926.81
  4793.1 1924.22  4856.7 1922.03  4913.3 1921.21  4969.8 1921.95  4976.8 1921.46
  4978.2 1919.86  4978.7 1919.36  4989.7 1919.86  5019.1 1922.34  5062.0 1921.45
  5175.2 1921.80  5246.7 1920.71  5445.7 1920.31  5651.3 1923.07  5999.7 1924.35
#Mann=3,-1,0
  4630.8    0.05       0  4978.2    0.05       0  4989.7    0.05       0
Bank Sta=4978.2,4989.7
Exp/Cntr=0.3,0.1

Type RM Length L Ch R = 1,160318,466,466,466
BEGIN DESCRIPTION:
Cedar Creek 160317.64
END DESCRIPTION:
XS GIS Cut Line= 4
      1574600.25      6774281.30      1574711.36      6774493.10
      1575292.07      6775200.79      1575762.54      6775243.14
#Sta/Elev= 30
  4763.8 1931.72  4771.4 1933.79  4780.9 1929.08  4786.5 1927.65  4793.9 1923.25
  4803.0 1921.83  4830.7 1920.92  4896.8 1920.81  4957.3 1921.28  4963.3 1921.17
  4979.4 1919.34  4985.9 1919.32  5016.2 1920.85  5059.2 1920.46  5065.7 1921.21
  5073.6 1920.60  5080.1 1921.18  5129.6 1921.29  5407.3 1919.93  5465.3 1919.04
  5465.8 1918.54  5476.4 1918.54  5476.9 1919.04  5513.8 1919.28  5527.1 1920.06
  5535.0 1919.65  5570.2 1919.47  5804.8 1921.74  6011.7 1923.09  6390.8 1924.39
#Mann=3,-1,0
  4763.8    0.05       0  5465.3   0.035       0  5476.9    0.05       0
Bank Sta=5465.3,5476.9
Exp/Cntr=0.3,0.1

Type RM Length L Ch R = 1,159852,264,264,264
BEGIN DESCRIPTION:
Cedar Creek 159851.99
END DESCRIPTION:
XS GIS Cut Line= 5
      1574183.50      6774765.93      1574412.66      6774786.77
      1574730.76      6774835.53      1575297.09      6775251.74
      1575770.17      6775310.82
#Sta/Elev= 30
  4769.5 1925.26  4846.9 1926.08  4931.7 1926.46  4941.7 1925.93  4951.7 1924.46
  4957.4 1920.97  4962.4 1918.57  4971.8 1918.67  4998.3 1920.00  5044.1 1920.76
  5123.4 1919.83  5327.1 1920.04  5404.5 1919.65  5534.1 1920.08  5548.7 1919.99
  5562.5 1919.44  5563.8 1917.52  5564.3 1917.02  5574.9 1917.02  5575.4 1917.52
  5575.8 1918.03  5584.2 1919.61  5590.4 1920.12  5634.4 1918.97  5669.9 1919.86
  5720.0 1919.86  6072.5 1923.07  6183.4 1923.25  6284.2 1923.97  6501.0 1924.19
#Mann=3,-1,0
  4769.5    0.05       0  5563.8    0.05       0  5575.4    0.05       0
Bank Sta=5563.8,5575.4
Exp/Cntr=0.3,0.1

Type RM Length L Ch R = 1,159588,602,602,602
BEGIN DESCRIPTION:
Cedar Creek 159587.54
END DESCRIPTION:
XS GIS Cut Line= 5
      1574092.32      6774953.43      1574355.37      6775000.31
      1574658.84      6775024.32      1575331.37      6775334.58
      1575957.91      6775469.70
#Sta/Elev= 30
  4732.2 1921.99  4775.5 1921.82  4795.9 1921.03  4896.6 1921.09  5001.7 1920.27
  5009.1 1919.19  5019.1 1916.94  5023.0 1916.83  5023.5 1916.33  5034.1 1916.33
  5034.6 1916.83  5039.1 1919.63  5049.2 1920.28  5059.2 1920.37  5162.4 1918.89
  5325.8 1919.16  5440.6 1920.06  5463.5 1919.61  5469.0 1916.99  5475.8 1917.01
  5492.0 1919.95  5497.8 1920.49  5552.9 1919.93  5596.9 1918.78  5718.1 1920.35
  5870.2 1921.42  5950.0 1922.51  6263.0 1923.73  6369.7 1923.32  6685.4 1925.75
#Mann=3,-1,0
  4732.2    0.05       0  5023.0    0.05       0  5034.6    0.05       0
Bank Sta=5023,5034.6
Exp/Cntr=0.3,0.1

Type RM Length L Ch R = 1,158986,830,830,830
BEGIN DESCRIPTION:
Mapping XS 4c7f0ceb
END DESCRIPTION:
XS GIS Cut Line= 4
      1573922.79      6774975.37      1574019.14      6775126.40
      1574224.87      6775504.01      1576438.84      6775538.28
#Sta/Elev= 30
  4524.2 1921.65  4550.7 1921.27  4629.4 1918.44  4665.7 1918.04  4805.8 1917.91
  4871.3 1917.15  4877.0 1917.76  4898.9 1917.53  4915.0 1918.38  4944.3 1918.04
  4989.9 1918.95  4996.7 1916.99  5002.4 1916.23  5018.5 1918.81  5153.5 1917.03
  5173.5 1914.85  5187.7 1914.36  5188.2 1913.86  5198.8 1913.86  5199.3 1914.36
  5213.5 1915.28  5223.5 1917.10  5333.5 1918.30  5633.6 1918.04  5853.6 1920.10
  6213.6 1921.50  6973.7 1927.06  7223.7 1928.26  7323.8 1929.42  7347.6 1930.29
#Mann=3,-1,0
  4524.2    0.05       0  5187.7    0.05       0  5199.3    0.05       0
Bank Sta=5187.7,5199.3
Exp/Cntr=0.3,0.1

Type RM Length L Ch R = 1,158156,438,438,438
BEGIN DESCRIPTION:
Cedar Creek 159255.76
END DESCRIPTION:
XS GIS Cut Line= 3
      1572054.74      6774918.07      1573766.53      6775633.35
      1576454.03      6775577.79
#Sta/Elev= 30
  3417.9 1918.85  3686.9 1917.79  3754.2 1915.91  3893.6 1917.29  3952.0 1914.22
  3960.1 1916.32  3975.8 1914.89  4014.3 1917.94  4058.1 1915.42  4264.8 1916.45
  4274.4 1914.21  4360.0 1916.30  4884.9 1915.51  4961.8 1915.63  4985.6 1917.12
  5000.5 1915.44  5003.5 1912.46  5004.0 1911.96  5015.2 1912.46  5022.2 1916.64
  5168.5 1915.19  5250.7 1916.14  5272.7 1915.91  5281.6 1914.09  5301.6 1916.24
  5631.7 1917.18  5661.7 1915.82  5681.7 1917.14  6181.8 1918.33  7961.2 1929.89
#Mann=3,-1,0
  3417.9    0.05       0  5003.5    0.05       0  5015.2    0.05       0
Bank Sta=5003.5,5015.2
Exp/Cntr=0.3,0.1

Type RM Length L Ch R = 1,157718,385,385,385
BEGIN DESCRIPTION:
Cedar Creek 159048.17
END DESCRIPTION:
XS GIS Cut Line= 3
      1571422.82      6775813.90      1573532.16      6775793.07
      1576260.68      6775725.38
#Sta/Elev= 30
  3214.0 1930.15  3556.2 1926.15  3606.2 1923.17  3816.2 1923.46  3926.2 1920.73
  3956.2 1916.34  4016.2 1914.41  4076.2 1913.22  4096.2 1916.59  4126.2 1913.45
  4176.2 1916.36  4266.2 1914.85  4280.4 1911.76  4280.9 1911.26  4292.1 1911.76
  4296.2 1915.21  4406.2 1912.51  4476.2 1916.08  4916.3 1914.91  4936.3 1912.87
  4966.3 1915.62  5026.3 1915.75  5396.3 1914.07  5876.4 1916.00  5986.5 1913.74
  6076.5 1916.79  7947.1 1927.01  8017.1 1929.01  8047.1 1933.53  8052.8 1932.30
#Mann=3,-1,0
  3214.0    0.05       0  4280.4   0.035       0  4292.1    0.05       0
Bank Sta=4280.4,4292.1
Exp/Cntr=0.3,0.1
