HEC-RAS study Cedar Creek.prj: Cedar Creek Base Level Engineering

--- Cedar Creek.g01 (geometry) --- (continued)

Type RM Length L Ch R = 1,157333,846,846,846
BEGIN DESCRIPTION:
Cedar Creek 158517.36
END DESCRIPTION:
XS GIS Cut Line= 4
      1571167.88      6776178.25      1572862.29      6776081.03
      1574390.07      6776164.36      1576631.56      6776199.06
#Sta/Elev= 30
  3165.7 1937.72  3633.6 1933.79  3703.7 1929.90  4064.3 1930.64  4302.2 1914.14
  4515.0 1911.28  4555.1 1913.91  4965.8 1914.55  4979.5 1910.41  4980.0 1909.91
  4992.0 1910.41  4995.8 1914.18  5005.8 1914.91  5326.3 1915.82  5356.3 1911.76
  5406.4 1911.12  5456.5 1911.26  5496.5 1916.29  5526.6 1912.50  5637.7 1911.70
  5666.8 1915.06  5736.9 1912.06  6001.5 1912.44  6127.5 1915.96  6157.5 1913.25
  6167.5 1916.09  6257.7 1917.44  7398.0 1921.11  8298.1 1928.15  8634.7 1934.89
#Mann=3,-1,0
  3165.7    0.05       0  4979.5   0.035       0  4992.0    0.05       0
Bank Sta=4979.5,4992
Exp/Cntr=0.3,0.1

Type RM Length L Ch R = 1,156487,779,779,779
BEGIN DESCRIPTION:
Cedar Creek 158107.79
END DESCRIPTION:
XS GIS Cut Line= 3
      1570785.87      6776837.97      1573757.64      6776756.63
      1576737.34      6776567.13
#Sta/Elev= 30
  3030.8 1944.50  3340.0 1941.28  3380.1 1937.86  3630.2 1928.39  3660.2 1929.14
  3750.2 1923.34  3810.2 1923.99  3860.2 1920.74  3990.3 1918.33  4600.5 1911.57
  4910.6 1912.25  4950.6 1910.15  4970.7 1912.55  4990.7 1911.68  4991.1 1909.76
  4991.6 1909.26  5010.3 1909.76  5010.7 1911.85  5020.7 1913.11  5092.6 1912.61
  5330.8 1912.13  5380.8 1909.83  5410.8 1912.16  5590.9 1912.76  5630.9 1910.93
  6151.3 1911.09  6472.0 1915.74  7123.3 1916.12  8295.7 1925.90  8989.4 1935.26
#Mann=4,-1,0
  3030.8    0.05       0  4991.1    0.07       0  5010.3    0.05       0
  5092.6    0.05       0
Bank Sta=4991.1,5010.3
Exp/Cntr=0.3,0.1

Type RM Length L Ch R = 1,155708,978,978,978
BEGIN DESCRIPTION:
Cedar Creek 157796.45
END DESCRIPTION:
XS GIS Cut Line= 3
      1570876.15      6777115.75      1573945.62      6777254.64
      1576674.74      6777310.19
#Sta/Elev= 30
  2818.8 1946.71  3158.0 1942.75  3358.2 1928.25  3388.2 1928.56  3448.3 1922.17
  3478.3 1923.11  3558.4 1918.07  3588.4 1918.91  3643.2 1916.12  3978.8 1912.22
  4539.4 1911.97  4559.4 1909.51  4589.5 1911.72  4619.5 1909.77  4689.6 1911.73
  4959.8 1911.34  4980.3 1909.48  4980.8 1908.98  4999.5 1909.48  4999.9 1911.08
  5029.9 1911.60  5830.7 1909.92  6140.8 1914.55  7601.1 1920.78  7711.2 1923.62
  7841.2 1923.00  8381.3 1928.67  8411.3 1931.39  8481.3 1930.06  8621.1 1935.42
#Mann=3,-1,0
  2818.8    0.05       0  4980.3    0.05       0  4999.5    0.05       0
Bank Sta=4980.3,4999.5
Exp/Cntr=0.3,0.1

Type RM Length L Ch R = 1,154730,1192,1192,1192
BEGIN DESCRIPTION:
Cedar Creek 159284.224
END DESCRIPTION:
XS GIS Cut Line= 3
      1570410.93      6777962.97      1573473.40      6778060.19
      1576445.62      6777949.08
#Sta/Elev= 30
  2353.9 1957.25  2666.5 1949.85  2978.3 1932.63  3288.4 1921.28  3648.6 1916.64
  3678.6 1920.81  3708.6 1916.44  4008.8 1913.32  4148.9 1915.71  4228.9 1911.75
  4549.1 1907.66  4739.2 1909.59  4859.2 1907.07  4875.2 1909.72  4959.3 1909.73
  4969.3 1909.61  4969.7 1905.25  4970.2 1904.75  4988.9 1905.25  4989.3 1908.12
  4999.3 1910.22  5052.6 1909.65  5151.6 1909.58  5209.4 1907.33  5299.4 1909.80
  7180.7 1915.30  7601.0 1918.97  7661.1 1921.79  8121.4 1923.25  8392.2 1932.84
#Mann=5,-1,0
  2353.9    0.05       0  4969.7    0.05       0  4988.9    0.05       0
  5052.6    0.12       0  5151.6    0.05       0
Bank Sta=4969.7,4988.9
Exp/Cntr=0.3,0.1

Type RM Length L Ch R = 1,153538,1162,1162,1162
BEGIN DESCRIPTION:
Cedar Creek 153538.49
END DESCRIPTION:
XS GIS Cut Line= 3
      1570398.25      6779143.85      1573148.28      6779050.10
      1576480.85      6778873.06
#Sta/Elev= 30
  2240.6 1943.41  2817.7 1932.37  2997.8 1931.90  3037.8 1928.25  3488.1 1921.02
  3828.3 1917.17  3958.3 1918.55  3988.4 1913.69  4728.8 1907.27  4768.8 1903.89
  4788.8 1907.10  5009.0 1907.88  5029.0 1904.21  5049.0 1907.75  5409.5 1907.36
  5619.8 1906.59  5638.8 1902.12  5639.3 1901.62  5660.9 1902.12  5679.9 1908.85
  5710.0 1905.36  6150.6 1905.54  6741.4 1909.02  6791.5 1911.50  7392.7 1912.96
  7432.4 1918.43  7462.4 1914.15  7672.7 1916.52  8073.3 1925.84  8329.5 1939.55
#Mann=3,-1,0
  2240.6    0.05       0  5638.8   0.035       0  5660.9    0.05       0
Bank Sta=5638.8,5660.9
Exp/Cntr=0.3,0.1

Type RM Length L Ch R = 1,152376,1800,1800,1800
BEGIN DESCRIPTION:
Cedar Creek 152375.75
END DESCRIPTION:
XS GIS Cut Line= 3
      1568761.35      6780619.29      1573296.97      6779968.25
      1576821.71      6778992.17
#Sta/Elev= 30
   409.4 2001.11   493.9 1997.45   797.0 2002.91  1484.0 1971.80  1645.4 1974.57
  2774.1 1942.42  2920.3 1949.35  3049.8 1945.87  3080.1 1937.06  3140.8 1932.24
  4100.5 1913.05  4151.0 1917.39  4282.3 1909.57  4878.4 1905.83  4996.5 1898.35
  4997.0 1897.85  5019.6 1898.35  5052.8 1905.73  5114.0 1900.98  5217.7 1906.91
  5308.4 1900.44  5500.7 1904.88  5540.2 1898.79  5560.2 1905.01  7484.6 1911.36
  7518.9 1918.31  7597.9 1913.13  7898.2 1920.65  8226.9 1938.35  8648.9 1940.85
#Mann=3,-1,0
   409.4    0.05       0  4996.5    0.05       0  5019.6    0.05       0
Bank Sta=4996.5,5019.6
Exp/Cntr=0.3,0.1

Type RM Length L Ch R = 1,150576,771,771,771
BEGIN DESCRIPTION:
Cedar Creek 150576.33
END DESCRIPTION:
XS GIS Cut Line= 3
      1569951.07      6781483.00      1574576.05      6780649.67
      1576930.14      6779149.72
#Sta/Elev= 30
   308.2 2017.39   515.4 2012.66   820.5 1992.04  1741.2 1949.23  1846.5 1944.95
  1902.1 1937.87  1996.9 1942.65  2173.0 1937.72  2333.8 1938.54  3279.2 1914.89
  4145.5 1902.90  4163.2 1899.79  4183.5 1903.19  4945.6 1900.11  4965.9 1899.33
  4978.4 1893.21  4978.9 1892.71  5001.9 1893.21  5004.6 1898.41  5037.4 1901.87
  6441.2 1910.16  6601.6 1915.13  6643.9 1923.44  6753.1 1918.90  6883.4 1924.58
  6977.4 1933.47  7354.2 1941.87  7477.6 1942.97  7701.9 1937.15  7799.0 1941.26
#Mann=5,-1,0
   308.2    0.05       0  1741.2    0.12       0  1902.1    0.05       0
  4978.4    0.05       0  5001.9    0.05       0
Bank Sta=4978.4,5001.9
Exp/Cntr=0.3,0.1

Type RM Length L Ch R = 1,149805,888,888,888
BEGIN DESCRIPTION:
Cedar Creek 149804.84
END DESCRIPTION:
XS GIS Cut Line= 3
      1570295.48      6781689.60      1574956.96      6781255.57
      1576471.43      6780923.47
#Sta/Elev= 30
   321.1 2013.41   503.3 1999.25   581.7 1988.12   612.5 1991.03   672.1 1983.93
   716.6 1990.02   929.9 1972.82  1314.9 1958.21  1366.6 1948.98  1515.8 1954.13
  2931.9 1916.90  3835.8 1899.78  3940.2 1902.55  4369.5 1900.71  4511.8 1899.66
  4601.6 1900.15  4619.1 1894.90  4649.3 1901.09  4715.9 1900.87  4930.5 1896.45
  4970.6 1900.60  4978.9 1890.66  4979.4 1890.16  5002.5 1890.66  5002.7 1894.34
  5031.5 1900.45  5420.5 1901.19  6300.9 1914.17  6460.8 1928.95  6553.2 1929.12
#Mann=7,-1,0
   321.1    0.05       0  3940.2    0.12       0  4369.5    0.05       0
  4511.8    0.12       0  4715.9    0.05       0  4978.9    0.05       0
  5002.5    0.05       0
Bank Sta=4978.9,5002.5
Exp/Cntr=0.3,0.1

Type RM Length L Ch R = 1,148917,1000,1000,1000
BEGIN DESCRIPTION:
Cedar Creek 148916.62
END DESCRIPTION:
XS GIS Cut Line= 4
      1570082.95      6782003.84      1574957.99      6781920.51
      1576160.57      6781960.19      1576281.01      6781887.25
#Sta/Elev= 30
   127.7 2053.52   219.8 2033.96   269.8 2032.74   309.8 2015.71   349.8 2022.03
   409.8 2015.29   599.8 2021.53   699.8 1994.37   789.8 1988.79   859.9 1969.91
  1099.9 1962.45  1229.9 1969.04  3170.2 1910.44  3990.3 1896.79  4133.5 1899.75
  4550.4 1899.15  4620.4 1892.36  4680.4 1898.65  4960.5 1898.79  4970.5 1897.08
  4978.7 1887.28  4979.2 1886.78  5002.3 1887.28  5040.5 1897.87  5077.5 1898.27
  5110.5 1893.38  5618.3 1898.98  5823.7 1903.32  6131.1 1909.03  6347.5 1927.19
#Mann=7,-1,0
   127.7    0.05       0  4133.5    0.12       0  4978.7    0.07       0
  5002.3    0.12       0  5077.5    0.05       0  5618.3    0.12       0
  5823.7    0.05       0
Bank Sta=4978.7,5002.3
Exp/Cntr=0.3,0.1

Type RM Length L Ch R = 1,147917,1486,1486,1486
BEGIN DESCRIPTION:
Cedar Creek 147917.02
END DESCRIPTION:
XS GIS Cut Line= 3
      1571035.07      6782870.30      1575207.45      6782731.26
      1580020.29      6782770.33
#Sta/Elev= 30
   825.3 1999.72  1105.4 1981.17  2055.9 1946.00  2548.5 1932.50  2726.3 1925.34
  2806.3 1917.00  3176.5 1911.71  3206.6 1905.83  3713.5 1898.79  3976.1 1895.99
  4154.0 1896.44  4285.7 1895.13  4518.5 1894.70  4977.5 1897.18  4995.7 1887.10
  4996.2 1886.60  5019.4 1887.10  5057.5 1897.03  5212.5 1896.36  5237.6 1893.38
  5914.7 1902.27  5961.0 1902.53  6337.6 1907.37  6707.6 1904.76  8647.7 1934.98
  8877.7 1941.94  8937.7 1948.47  9047.7 1949.00  9727.7 1983.06  9813.0 1991.86
#Mann=11,-1,0
   825.3    0.05       0  3713.5    0.12       0  3976.1    0.05       0
  4154.0    0.12       0  4285.7    0.05       0  4518.5    0.12       0
  4995.7    0.07       0  5019.4    0.12       0  5212.5    0.05       0
  5914.7    0.12       0  5961.0    0.05       0
Bank Sta=4995.7,5019.4
Exp/Cntr=0.3,0.1

Type RM Length L Ch R = 1,146431,1057,1057,1057
BEGIN DESCRIPTION:
Cedar Creek 146430.52
END DESCRIPTION:
XS GIS Cut Line= 3
      1571616.64      6784207.11      1575210.41      6783920.65
      1579575.60      6783735.18
#Sta/Elev= 30
  1400.6 1977.55  1827.6 1958.45  2261.7 1945.84  2458.2 1932.56  2472.4 1936.34
  2502.4 1933.90  2663.0 1938.89  2965.7 1927.87  3134.4 1914.57  3244.8 1917.17
  4447.0 1892.92  4589.0 1892.73  4619.1 1887.02  4649.2 1891.92  4772.8 1892.28
  4980.7 1893.06  5008.5 1883.94  5009.0 1883.44  5032.3 1883.94  5040.4 1892.76
  5049.8 1892.95  5122.1 1892.48  6862.0 1904.07  7539.6 1912.42  8283.3 1930.21
  8693.7 1935.74  8952.0 1950.85  9064.0 1950.61  9094.0 1955.18  9374.9 1964.73
#Mann=7,-1,0
  1400.6    0.05       0  4447.0    0.12       0  4772.8    0.05       0
  5008.5    0.05       0  5032.3    0.05       0  5049.8    0.12       0
  5122.1    0.05       0
Bank Sta=5008.5,5032.3
Exp/Cntr=0.3,0.1

Type RM Length L Ch R = 1,145374,3038,3038,3038
BEGIN DESCRIPTION:
Cedar Creek 145373.5
END DESCRIPTION:
XS GIS Cut Line= 3
      1571885.80      6785109.88      1575557.64      6784745.30
      1579191.81      6784424.57
#Sta/Elev= 30
  1312.6 1969.00  1663.5 1954.39  2939.8 1923.60  3110.6 1913.73  3693.5 1900.74
  3954.7 1899.83  3994.9 1896.04  4607.9 1888.80  4859.2 1890.80  4919.5 1885.68
  4949.6 1890.04  4969.7 1888.38  4977.3 1883.43  4977.8 1882.93  5002.2 1883.43
  5002.5 1888.76  5040.0 1890.81  5090.2 1890.67  5130.4 1885.55  5160.5 1891.35
  5597.3 1894.99  5702.6 1887.60  5821.5 1898.83  5903.3 1893.00  6050.7 1897.00
  6174.4 1894.96  6636.2 1906.56  7158.2 1909.72  8001.5 1927.37  8650.8 1949.47
#Mann=3,-1,0
  1312.6    0.05       0  4977.3    0.05       0  5002.2    0.05       0
Bank Sta=4977.3,5002.2
Exp/Cntr=0.3,0.1

Type RM Length L Ch R = 1,142336,1882,1882,1882
BEGIN DESCRIPTION:
Cedar Creek 142239.73
END DESCRIPTION:
XS GIS Cut Line= 3
      1571589.47      6786274.13      1576658.91      6786121.35
      1580560.81      6785947.78
#Sta/Elev= 30
   -68.0 1990.03   -29.1 1981.10    57.7 1981.62   429.3 1961.55   507.8 1965.12
  1288.1 1932.50  2088.5 1914.79  3291.5 1903.48  4049.4 1888.19  4849.8 1885.12
  4885.4 1874.99  4885.9 1874.49  4914.2 1874.99  4939.8 1886.07  4979.8 1883.65
  4989.8 1877.11  5029.9 1891.90  5119.9 1887.16  6501.3 1899.82  7302.1 1931.77
  7532.3 1947.39  7772.6 1951.89  8002.8 1980.69  8094.7 2000.58  8363.1 2042.95
  8423.2 2042.28  8483.3 2065.18  8567.6 2081.12  8683.5 2146.31  8909.5 2218.04
#Mann=7,-1,0
   -68.0    0.05       0    57.7    0.12       0   429.3    0.05       0
  4885.4    0.07       0  4914.2    0.05       0  5119.9    0.05       0
  8094.7    0.12       0
Bank Sta=4885.4,4914.2
Exp/Cntr=0.3,0.1

Type RM Length L Ch R = 1,140454,2010,2010,2010
BEGIN DESCRIPTION:
Cedar Creek 140454.2
END DESCRIPTION:
XS GIS Cut Line= 4
      1573186.07      6787873.99      1576451.73      6787733.37
      1577206.94      6787389.62      1580611.29      6786093.47
#Sta/Elev= 30
   891.1 1939.98  2351.4 1910.03  2941.9 1907.32  3232.2 1893.88  3392.4 1897.66
  3542.5 1885.56  4153.1 1878.50  4981.7 1883.00  4998.4 1872.68  4998.7 1872.18
  5012.8 1872.68  5060.7 1882.18  5112.2 1881.41  5141.4 1881.35  5236.0 1882.19
  5276.4 1875.13  5308.5 1880.91  5733.3 1883.26  5889.3 1885.99  7216.2 1932.29
  7317.6 1939.66  7445.7 1949.40  7757.9 1968.11  7881.9 1983.95  8068.2 2013.73
  8347.3 2068.90  8467.7 2116.17  8572.1 2147.34  8614.9 2169.29  8632.3 2187.05
#Mann=12,-1,0
   891.1    0.05       0  4998.4    0.05       0  5012.8    0.05       0
  5112.2    0.12       0  5141.4    0.05       0  5733.3    0.12       0
  5889.3    0.05       0  7216.2   0.075       0  7317.6    0.05       0
  7445.7    0.12       0  7881.9    0.05       0  8068.2    0.12       0
Bank Sta=4998.4,5012.8
Exp/Cntr=0.3,0.1

Type RM Length L Ch R = 1,138444,1074,1074,1074
BEGIN DESCRIPTION:
Cedar Creek 138444.4
END DESCRIPTION:
XS GIS Cut Line= 3
      1573272.82      6788422.06      1577054.09      6788474.14
      1579944.76      6787989.76
#Sta/Elev= 30
  1216.7 1936.16  1355.4 1933.39  1450.9 1929.54  1751.2 1925.70  2859.0 1905.77
  3079.1 1910.29  3169.1 1899.80  3299.1 1896.33  3339.1 1900.76  3369.1 1893.52
  3679.1 1892.26  3969.1 1883.66  4709.2 1875.07  4759.2 1878.03  4819.2 1872.59
  4989.2 1877.30  4996.3 1873.97  4997.5 1868.62  4997.7 1868.12  5012.4 1868.62
  5039.8 1878.08  5070.5 1878.44  5333.9 1879.28  5404.8 1873.61  5475.8 1880.25
  5769.9 1880.30  6023.3 1875.04  7562.0 1926.49  7638.2 1930.20  7929.3 1942.67
#Mann=8,-1,0
  1216.7    0.12       0  1355.4    0.05       0  1450.9    0.12       0
  1751.2    0.05       0  4997.5    0.05       0  5012.4    0.05       0
  7562.0    0.12       0  7638.2    0.05       0
Bank Sta=4997.5,5012.4
Exp/Cntr=0.3,0.1

Type RM Length L Ch R = 1,137370,1290,1290,1290
BEGIN DESCRIPTION:
Mapping XS e2f91981
END DESCRIPTION:
XS GIS Cut Line= 4
      1573933.44      6789137.58      1576502.92      6789248.69
      1578655.70      6789116.75      1579231.03      6788991.98
#Sta/Elev= 30
  1273.6 1917.70  1565.4 1910.18  2266.1 1907.74  2496.3 1903.64  2789.7 1904.39
  2886.7 1902.53  2956.7 1894.07  3056.8 1891.10  3126.9 1890.55  3176.9 1894.78
  3207.0 1892.79  3251.4 1895.25  3387.1 1888.94  3601.3 1883.60  3835.4 1880.88
  4979.7 1876.12  4989.7 1871.88  4992.4 1866.80  4992.7 1866.30  5007.4 1866.80
  5019.8 1872.23  5049.8 1878.32  5245.7 1875.04  5420.5 1877.61  5440.5 1872.38
  5460.6 1877.86  5851.3 1877.41  6482.5 1892.39  6564.4 1895.11  6591.0 1898.35
#Mann=5,-1,0
  1273.6    0.05       0  3601.3    0.12       0  3835.4    0.05       0
  4992.4    0.05       0  5007.4    0.05       0
Bank Sta=4992.4,5007.4
Exp/Cntr=0.3,0.1

Type RM Length L Ch R = 1,136080,1704,1704,1704
BEGIN DESCRIPTION:
Cedar Creek 137377.38
END DESCRIPTION:
XS GIS Cut Line= 3
      1575329.34      6791588.95      1576793.68      6790359.56
      1579246.76      6789963.73
#Sta/Elev= 30
  1748.9 1911.64  1945.2 1907.13  2265.2 1908.55  2306.9 1905.17  2485.0 1910.63
  2555.3 1896.99  2612.5 1892.23  3130.3 1882.28  3272.1 1880.83  3315.0 1883.85
  3343.6 1880.80  3655.8 1881.65  4472.6 1873.78  4503.0 1873.00  4533.4 1867.51
  4543.5 1871.55  4573.9 1873.86  4915.4 1873.20  4979.0 1874.06  4985.8 1871.45
  4997.3 1864.82  4997.5 1864.32  5012.2 1864.82  5017.4 1870.86  5029.7 1874.80
  5252.5 1870.06  5323.4 1874.06  5393.1 1870.17  6062.9 1879.87  6145.7 1884.72
#Mann=5,-1,0
  1748.9    0.05       0  4915.4    0.12       0  4985.8    0.05       0
  4997.3    0.05       0  5012.2    0.05       0
Bank Sta=4997.3,5012.2
Exp/Cntr=0.3,0.1

Type RM Length L Ch R = 1,134376,1505,1505,1505
BEGIN DESCRIPTION:
Cedar Creek 134376.09
END DESCRIPTION:
XS GIS Cut Line= 3
      1575547.23      6792050.50      1578026.37      6791001.90
      1579257.82      6790409.07
#Sta/Elev= 30
  2314.4 1919.48  2648.6 1916.93  2871.9 1906.08  2909.2 1902.06  2972.1 1905.51
  3148.0 1902.14  3201.7 1897.17  3213.2 1891.79  3236.2 1888.28  3354.3 1883.22
  3886.3 1873.51  4442.1 1873.82  4571.4 1872.95  4635.5 1869.93  4666.2 1872.87
  4948.5 1871.90  4972.1 1862.37  4978.1 1862.37  4978.3 1861.87  4994.1 1862.37
  5001.3 1869.91  5024.0 1871.31  5493.2 1871.57  5570.7 1870.65  5583.7 1867.08
  5615.1 1871.00  5748.3 1868.00  5781.6 1870.37  6335.9 1875.26  6372.9 1879.28
#Mann=3,-1,0
  2314.4    0.05       0  4978.1    0.05       0  4994.1    0.05       0
Bank Sta=4978.1,4994.1
Exp/Cntr=0.3,0.1

Type RM Length L Ch R = 1,132871,1861,1861,1861
BEGIN DESCRIPTION:
Cedar Creek 132871.05
END DESCRIPTION:
XS GIS Cut Line= 3
      1575692.99      6792814.42      1578151.37      6791897.73
      1579277.27      6791360.80
#Sta/Elev= 30
  2365.8 1904.07  2496.1 1900.97  2683.7 1894.75  2868.2 1894.40  3600.6 1881.15
  3661.3 1873.97  3691.6 1877.93  4096.9 1875.25  4139.3 1879.03  4175.0 1872.70
  4395.7 1871.70  4431.9 1879.17  4487.2 1869.90  4663.7 1868.42  4737.3 1873.16
  4790.6 1868.52  4865.3 1869.20  4874.1 1861.41  4874.6 1860.91  4906.4 1861.41
  4950.9 1866.28  5045.2 1863.22  5060.0 1868.06  5126.5 1869.35  5674.6 1869.64
  5702.8 1862.51  5735.8 1869.37  5856.1 1870.54  6088.6 1865.16  6236.9 1873.03
#Mann=5,-1,0
  2365.8    0.05       0  2496.1    0.12       0  2868.2    0.05       0
  4874.1    0.05       0  4906.4    0.05       0
Bank Sta=4874.1,4906.4
Exp/Cntr=0.3,0.1

Type RM Length L Ch R = 1,131010,863,863,863
BEGIN DESCRIPTION:
Cedar Creek 131009.6
END DESCRIPTION:
XS GIS Cut Line= 3
      1575962.42      6794014.05      1578899.89      6792472.40
      1579359.86      6792213.45
#Sta/Elev= 30
  1690.0 1908.44  1772.0 1908.28  1966.4 1894.39  1999.5 1893.56  2273.9 1887.31
  2483.1 1888.31  2607.7 1881.03  2957.0 1882.02  3265.8 1875.77  3533.8 1879.08
  3734.0 1873.47  3838.6 1879.03  3917.7 1869.97  4097.6 1869.18  4147.3 1873.42
  4555.0 1864.04  4577.1 1867.75  4956.7 1867.61  4968.4 1866.51  4984.3 1856.63
  4984.5 1856.13  5000.6 1856.63  5001.2 1861.86  5006.8 1866.35  5036.3 1867.58
  5374.0 1867.55  5395.6 1866.30  5403.5 1861.20  5449.2 1868.49  5535.3 1869.81
#Mann=5,-1,0
  1690.0    0.05       0  1966.4    0.12       0  1999.5    0.05       0
  4984.3    0.05       0  5000.6    0.05       0
Bank Sta=4984.3,5000.6
Exp/Cntr=0.3,0.1

Type RM Length L Ch R = 1,130147,1380,1380,1380
BEGIN DESCRIPTION:
Cedar Creek 130147.35
END DESCRIPTION:
XS GIS Cut Line= 3
      1576406.81      6794521.03      1579302.67      6793041.84
      1579424.21      6792992.34
#Sta/Elev= 30
  1745.6 1914.62  1872.9 1900.12  2013.1 1891.16  2384.0 1879.10  2839.4 1874.83
  2972.7 1879.36  2989.4 1874.97  3078.2 1873.70  3225.8 1873.90  3270.7 1879.05
  3315.6 1873.18  3439.4 1872.59  3522.6 1872.62  3567.1 1878.94  3605.9 1870.90
  3656.0 1868.20  3820.9 1867.84  3865.9 1873.43  3894.8 1867.51  4405.9 1865.60
  4466.9 1860.89  4489.1 1865.68  4943.8 1865.80  4966.3 1863.86  4990.5 1854.96
  4990.8 1854.46  5006.9 1854.96  5032.3 1865.04  5047.9 1861.78  5128.6 1869.54
#Mann=3,-1,0
  1745.6    0.05       0  4990.5    0.05       0  5006.9    0.05       0
Bank Sta=4990.5,5006.9
Exp/Cntr=0.3,0.1

Type RM Length L Ch R = 1,128767,734,734,734
BEGIN DESCRIPTION:
Cedar Creek 128559.27
END DESCRIPTION:
XS GIS Cut Line= 3
      1579600.37      6794019.96      1579789.38      6793916.23
      1580997.72      6790166.21
#Sta/Elev= 30
  4512.5 1868.66  4540.6 1867.23  4563.1 1862.76  4597.6 1861.37  4896.4 1862.34
  4928.4 1868.31  4978.4 1855.97  4996.6 1853.46  4996.9 1852.96  5013.4 1853.46
  5062.5 1862.64  5409.2 1862.72  5451.9 1858.74  5516.1 1862.60  5612.3 1863.09
  5661.3 1860.41  6066.4 1866.79  6176.1 1866.29  6392.3 1869.45  6686.1 1870.53
  6883.7 1873.98  6995.6 1872.99  7058.7 1875.35  7153.2 1874.72  7615.5 1883.07
  8331.0 1899.14  8436.1 1901.98  8535.0 1906.03  8637.0 1911.38  8668.0 1912.51
#Mann=7,-1,0
  4512.5    0.05       0  4996.6    0.05       0  5013.4    0.05       0
  8331.0    0.12       0  8436.1    0.05       0  8535.0    0.12       0
  8637.0    0.05       0
Bank Sta=4996.6,5013.4
Exp/Cntr=0.3,0.1

Type RM Length L Ch R = 1,128033,824,824,824
BEGIN DESCRIPTION:
Mapping XS 7393c39e
END DESCRIPTION:
XS GIS Cut Line= 4
      1579629.67      6794443.98      1579643.55      6794423.17
      1581733.83      6793694.00      1582983.80      6792207.92
#Sta/Elev= 30
  4381.0 1868.38  4418.1 1868.16  4449.9 1861.68  4497.6 1859.39  4915.9 1860.28
  4937.1 1862.10  4986.4 1852.28  4986.8 1851.78  5003.7 1852.28  5040.9 1861.68
  5439.5 1859.86  5470.6 1860.53  5501.6 1864.75  5527.4 1858.13  5620.6 1858.25
  5636.1 1860.37  5646.4 1858.36  5699.7 1858.14  5739.6 1863.56  5770.6 1861.20
  6138.1 1864.64  6666.9 1872.98  6845.1 1879.38  6880.2 1883.67  6908.8 1881.76
  7221.0 1889.29  7654.1 1893.11  7966.2 1901.81  8286.2 1914.90  8561.7 1919.53
#Mann=3,-1,0
  4381.0    0.05       0  4986.4   0.035       0  5003.7    0.05       0
Bank Sta=4986.4,5003.7
Exp/Cntr=0.3,0.1

Type RM Length L Ch R = 1,127209,1044,1044,1044
BEGIN DESCRIPTION:
Cedar Creek 127208.89
END DESCRIPTION:
XS GIS Cut Line= 4
      1579709.95      6795168.04      1580226.72      6795008.50
      1581952.14      6794322.27      1582201.70      6793791.97
#Sta/Elev= 30
  4459.9 1868.43  4478.9 1867.98  4506.3 1861.42  4538.4 1858.50  4881.2 1858.82
  4919.1 1857.39  4946.5 1858.51  4983.6 1850.93  4983.9 1850.43  5000.9 1850.93
  5020.7 1856.62  5031.2 1857.92  5300.2 1856.33  5601.6 1857.24  5655.4 1858.96
  5859.8 1856.95  6354.9 1862.94  6507.4 1866.08  6537.8 1869.14  6548.6 1867.95
  6639.6 1871.34  6753.1 1885.67  6839.2 1888.15  7006.0 1887.41  7059.8 1882.86
  7337.6 1886.61  7359.7 1886.21  7381.8 1881.76  7390.0 1881.69  7443.7 1885.71
#Mann=3,-1,0
  4459.9    0.05       0  4983.6    0.05       0  5000.9    0.05       0
Bank Sta=4983.6,5000.9
Exp/Cntr=0.3,0.1

Type RM Length L Ch R = 1,126165,738,738,738
BEGIN DESCRIPTION:
Cedar Creek 126165.22
END DESCRIPTION:
XS GIS Cut Line= 4
      1579790.71      6795957.69      1580879.49      6795772.39
      1581457.35      6795598.31      1582139.63      6794374.38
#Sta/Elev= 30
  3887.5 1868.36  3902.0 1867.89  3932.4 1860.13  3962.9 1857.99  4409.2 1856.52
  4936.7 1857.19  4946.8 1857.07  4984.0 1850.49  4984.4 1849.99  5001.3 1850.49
  5008.1 1854.30  5018.6 1856.36  5057.1 1857.33  5217.0 1855.52  5435.8 1856.76
  5675.9 1856.67  5733.2 1855.43  5769.2 1856.41  5909.8 1855.59  6153.2 1858.09
  6402.4 1865.01  6527.0 1870.16  6602.4 1873.71  6608.1 1875.00  6624.1 1875.30
  6651.6 1878.44  6711.0 1882.59  6776.2 1885.84  6873.3 1886.74  6996.7 1883.07
#Mann=3,-1,0
  3887.5    0.05       0  4984.0    0.05       0  5001.3    0.05       0
Bank Sta=4984,5001.3
Exp/Cntr=0.3,0.1

Type RM Length L Ch R = 1,125427,1433,1433,1433
BEGIN DESCRIPTION:
Mapping XS 89c3d3b6
END DESCRIPTION:
XS GIS Cut Line= 4
      1579900.04      6796910.82      1580983.39      6796546.23
      1582233.39      6795681.65      1583951.03      6795161.15
#Sta/Elev= 30
  3335.3 1868.77  3372.2 1864.35  3484.1 1860.89  3899.7 1853.54  4392.4 1852.23
  4542.0 1854.24  4637.3 1852.61  4989.4 1854.38  4995.5 1853.99  4999.5 1846.11
  4999.9 1845.61  5017.0 1846.11  5025.2 1846.53  5031.3 1851.31  5039.6 1853.16
  5219.1 1854.43  5261.0 1851.76  5513.8 1854.83  5577.3 1850.40  5613.1 1854.72
  5830.0 1854.71  6020.8 1860.11  6858.8 1870.45  6950.8 1872.98  7023.4 1878.65
  7044.8 1877.36  7066.7 1880.33  7132.6 1882.56  7264.2 1884.10  7793.0 1897.32
#Mann=3,-1,0
  3335.3    0.05       0  4999.5    0.05       0  5017.0    0.05       0
Bank Sta=4999.5,5017
Exp/Cntr=0.3,0.1

Type RM Length L Ch R = 1,123994,2240,2240,2240
BEGIN DESCRIPTION:
Cedar Creek 124242.939
END DESCRIPTION:
XS GIS Cut Line= 3
      1579483.41      6797276.26      1582592.77      6796948.14
      1584415.67      6796708.56
#Sta/Elev= 30
  2462.8 1899.17  2565.0 1900.30  2665.5 1876.56  2806.3 1873.07  2846.5 1870.16
  2866.6 1865.74  2886.7 1868.32  2937.0 1865.12  2971.3 1867.54  3017.5 1863.44
  3278.9 1856.89  3630.8 1851.72  3729.5 1855.97  3771.6 1848.88  3811.8 1850.58
  3827.4 1854.54  4254.3 1848.05  4606.2 1852.13  4928.0 1851.49  4972.3 1850.13
  4985.2 1844.77  4985.7 1844.27  5003.1 1844.77  5008.4 1849.80  5018.5 1850.70
  5621.9 1852.00  5904.3 1861.92  6368.3 1872.13  6993.6 1876.08  7428.0 1883.01
#Mann=3,-1,0
  2462.8    0.05       0  4985.2    0.05       0  5003.1    0.05       0
Bank Sta=4985.2,5003.1
Exp/Cntr=0.3,0.1

Type RM Length L Ch R = 1,121754,919,919,919
BEGIN DESCRIPTION:
Cedar Creek 121753.65
END DESCRIPTION:
XS GIS Cut Line= 3
      1578752.66      6797548.59      1583153.75      6797835.05
      1586287.45      6797835.05
#Sta/Elev= 30
   588.6 1898.50   761.3 1897.68   921.6 1888.26  1422.0 1877.83  1833.6 1864.42
  2003.9 1864.05  2154.2 1857.78  2755.5 1849.61  3386.8 1848.11  3396.9 1847.88
  3406.1 1840.59  3407.0 1840.09  3443.7 1840.59  3527.1 1846.63  3607.3 1843.55
  3667.4 1848.19  4138.4 1849.04  4940.1 1846.58  4971.3 1845.64  4990.2 1841.09
  5080.2 1847.14  5130.2 1854.91  5200.2 1859.20  5410.2 1881.90  5760.2 1879.74
  5840.2 1886.30  6170.2 1901.48  7080.2 1910.85  7590.2 1909.26  8132.7 1919.77
#Mann=3,-1,0
   588.6    0.05       0  3406.1    0.05       0  3443.7    0.05       0
Bank Sta=3406.1,3443.7
Exp/Cntr=0.3,0.1

Type RM Length L Ch R = 1,120835,1720,1720,1720
BEGIN DESCRIPTION:
Cedar Creek 120835.38
END DESCRIPTION:
XS GIS Cut Line= 3
      1578787.38      6798069.42      1582954.09      6798651.02
      1586148.57      6798381.92
#Sta/Elev= 30
   790.2 1901.72   909.0 1904.32  1034.1 1901.79  1131.1 1894.80  1312.8 1892.58
  1363.3 1888.27  1383.5 1883.25  1484.5 1877.07  2140.8 1859.39  3241.4 1847.28
  3251.4 1846.50  3252.3 1837.10  3253.2 1836.60  3289.9 1837.10  3433.2 1837.10
  3443.3 1837.53  3463.5 1845.59  3544.3 1846.78  4079.4 1841.50  4935.9 1845.02
  5000.3 1837.31  5018.3 1842.71  5088.2 1845.40  5770.9 1853.69  6212.5 1873.70
  6383.1 1887.76  6483.5 1883.80  6624.0 1885.40  6804.6 1892.63  8203.1 1911.07
#Mann=3,-1,0
   790.2    0.05       0  3252.3    0.05       0  3289.9    0.05       0
Bank Sta=3252.3,3289.9
Exp/Cntr=0.3,0.1

Type RM Length L Ch R = 1,119115,1506,1506,1506
BEGIN DESCRIPTION:
Cedar Creek 119115.46
END DESCRIPTION:
XS GIS Cut Line= 3
      1578830.84      6799276.02      1583362.08      6799553.80
      1586224.81      6799102.71
#Sta/Elev= 30
   451.4 1896.00   575.8 1893.31   716.1 1881.82   891.8 1873.43  1136.8 1866.14
  1878.2 1855.20  2309.0 1851.85  2429.3 1854.31  2525.5 1849.33  3250.8 1842.30
  3531.3 1843.59  4032.3 1838.69  4072.3 1841.52  4102.4 1837.81  4192.6 1843.15
  4923.5 1843.20  4973.5 1837.94  4978.5 1841.00  4992.7 1832.37  4993.2 1831.87
  5011.6 1832.37  5044.7 1841.00  5166.2 1840.26  5185.2 1836.75  5224.3 1840.65
  5277.6 1854.34  5368.7 1865.21  5468.2 1868.23  5945.7 1884.02  7889.2 1899.47
#Mann=6,-1,0
   451.4    0.05       0  4923.5    0.12       0  4992.7    0.07       0
  5011.6    0.12       0  5224.3    0.12       0  5468.2    0.05       0
Bank Sta=4992.7,5011.6
Exp/Cntr=0.3,0.1

Type RM Length L Ch R = 1,117609,927,927,927
BEGIN DESCRIPTION:
Cedar Creek 117608.61
END DESCRIPTION:
XS GIS Cut Line= 3
      1578937.59      6800137.13      1584111.21      6800406.23
      1586324.77      6800215.26
#Sta/Elev= 30
  -174.5 1889.90   523.9 1865.02  1024.5 1858.91  1044.6 1862.61  1234.8 1861.44
  2126.0 1847.43  3748.2 1839.28  3786.0 1832.53  3848.3 1838.88  4048.6 1835.71
  4349.0 1842.18  4590.3 1840.96  4759.4 1839.50  4957.3 1835.46  5000.5 1829.26
  5001.0 1828.76  5019.5 1829.26  5056.6 1837.30  5157.8 1848.84  5431.5 1851.35
  5521.8 1866.43  5582.0 1868.54  5672.4 1865.56  5739.7 1852.74  5772.7 1853.35
  5822.9 1868.42  5863.1 1865.41  6104.0 1878.51  6375.0 1884.78  7227.9 1887.10
#Mann=7,-1,0
  -174.5    0.05       0  4590.3    0.12       0  4759.4    0.05       0
  4957.3    0.12       0  5000.5    0.07       0  5019.5    0.12       0
  5056.6    0.05       0
Bank Sta=5000.5,5019.5
Exp/Cntr=0.3,0.1

Type RM Length L Ch R = 1,116682,2112,2112,2112
BEGIN DESCRIPTION:
Cedar Creek 116682.23
END DESCRIPTION:
XS GIS Cut Line= 3
      1578790.07      6801031.23      1584406.35      6801083.32
      1586836.92      6800770.81
#Sta/Elev= 30
  -614.7 1884.73   180.3 1860.53   820.3 1859.35  1360.3 1849.68  1490.3 1853.26
  2310.4 1843.49  3590.4 1838.18  3630.4 1842.25  3780.4 1832.41  4243.2 1832.91
  4410.4 1832.04  4670.5 1829.49  4730.5 1837.25  4884.4 1837.48  4960.5 1834.97
  4985.8 1826.64  4986.3 1826.14  5004.8 1826.64  5020.6 1833.97  5089.5 1843.66
  5243.5 1849.17  5454.2 1846.96  5477.1 1852.85  5504.6 1847.32  5556.6 1847.39
  5636.2 1857.78  5817.1 1867.92  6059.1 1874.37  6462.4 1880.75  7452.4 1883.90
#Mann=7,-1,0
  -614.7    0.05       0  4243.2    0.12       0  4410.4    0.05       0
  4884.4    0.12       0  4985.8    0.07       0  5004.8    0.12       0
  5089.5    0.05       0
Bank Sta=4985.8,5004.8
Exp/Cntr=0.3,0.1

Type RM Length L Ch R = 1,114570,534,534,534
BEGIN DESCRIPTION:
Cedar Creek 114569.9
END DESCRIPTION:
XS GIS Cut Line= 3
      1578869.92      6801996.51      1583609.47      6801883.66
      1587610.57      6801883.66
#Sta/Elev= 30
   263.0 1874.01   598.2 1871.67   748.2 1866.90   768.2 1861.87   788.2 1866.08
   878.3 1865.49  2158.6 1849.35  3008.9 1844.56  3138.9 1847.44  3569.0 1841.48
  4819.4 1835.95  4939.4 1827.04  4959.4 1829.61  4980.0 1823.62  4980.5 1823.12
  4999.4 1823.62  5019.4 1830.12  5129.4 1833.55  5499.4 1833.00  6589.4 1842.97
  6979.4 1859.17  7339.4 1851.41  7369.4 1852.51  7389.4 1857.98  7489.4 1855.16
  7589.4 1864.78  7839.4 1870.55  8189.4 1862.29  8469.4 1871.93  9005.0 1875.42
#Mann=3,-1,0
   263.0    0.05       0  4980.0   0.035       0  4999.4    0.05       0
Bank Sta=4980,4999.4
Exp/Cntr=0.3,0.1

Type RM Length L Ch R = 1,114036,997,997,997
BEGIN DESCRIPTION:
Cedar Creek 114035.67
END DESCRIPTION:
XS GIS Cut Line= 3
      1579121.59      6802473.94      1583813.88      6802343.49
      1586290.87      6802298.86
#Sta/Elev= 30
   305.9 1868.60   779.5 1866.66  1709.9 1852.32  2370.1 1853.25  2980.3 1843.87
  3110.4 1845.80  3140.4 1843.02  3370.5 1839.86  4302.7 1837.06  4622.7 1835.98
  4871.1 1832.46  4951.1 1828.56  4989.3 1822.88  4989.8 1822.38  5008.8 1822.88
  5061.1 1831.77  5091.1 1831.74  5111.1 1828.05  5181.2 1828.03  5211.2 1834.11
  5392.5 1830.78  5642.3 1832.81  6351.3 1835.50  6641.4 1840.68  6689.4 1835.22
  6731.4 1841.18  6971.4 1843.25  7171.5 1853.26  7331.5 1865.55  7477.4 1864.69
#Mann=7,-1,0
   305.9    0.05       0  4302.7    0.12       0  4622.7    0.05       0
  4989.3   0.035       0  5008.8    0.05       0  5392.5    0.12       0
  5642.3    0.05       0
Bank Sta=4989.3,5008.8
Exp/Cntr=0.3,0.1

Type RM Length L Ch R = 1,113039,1398,1398,1398
BEGIN DESCRIPTION:
Cedar Creek 113038.63
END DESCRIPTION:
XS GIS Cut Line= 3
      1580806.52      6803310.60      1584200.62      6803197.75
      1587211.36      6802911.43
#Sta/Elev= 30
  1599.3 1875.89  1647.8 1880.53  1677.8 1887.09  1727.8 1883.77  1767.9 1887.87
  1857.9 1874.39  2008.0 1867.40  2058.0 1869.35  2078.0 1865.24  2298.2 1857.04
  2908.5 1849.00  3027.7 1851.96  3118.6 1847.07  4580.4 1830.72  4679.5 1831.63
  4929.6 1823.69  4939.6 1825.53  4985.0 1821.40  4985.5 1820.90  5004.7 1821.40
  5009.7 1825.84  5039.9 1827.70  5220.7 1830.08  5592.3 1826.51  6630.9 1833.09
  6928.3 1839.54  7229.7 1858.36  7320.1 1858.96  7390.4 1863.37  8019.6 1865.27
#Mann=5,-1,0
  1599.3    0.05       0  4580.4    0.12       0  4679.5    0.05       0
  4985.0   0.035       0  5004.7    0.05       0
Bank Sta=4985,5004.7
Exp/Cntr=0.3,0.1

Type RM Length L Ch R = 1,111641,1092,1092,1092
BEGIN DESCRIPTION:
Cedar Creek 111641.37
END DESCRIPTION:
XS GIS Cut Line= 3
      1581563.46      6804463.38      1584705.83      6804072.75
      1587917.66      6803664.76
#Sta/Elev= 30
  1833.6 1861.84  1946.0 1857.77  2117.3 1863.10  2404.3 1862.53  2802.5 1851.38
  2852.9 1852.77  2873.1 1849.87  2913.4 1852.53  2943.6 1849.51  3034.3 1848.12
  3790.1 1839.32  3971.5 1832.53  4898.6 1827.29  4974.7 1818.70  4975.2 1818.20
  4994.4 1818.70  4996.2 1822.94  4999.2 1823.62  5019.5 1824.03  5110.2 1822.14
  5463.0 1827.29  5854.2 1827.20  5956.0 1827.51  6271.2 1827.36  6491.2 1831.79
  6906.2 1855.41  6954.9 1855.32  7066.1 1848.88  7166.6 1858.46  8237.8 1859.44
#Mann=5,-1,0
  1833.6    0.05       0  4974.7   0.035       0  4994.4    0.05       0
  5854.2    0.12       0  5956.0    0.05       0
Bank Sta=4974.7,4994.4
Exp/Cntr=0.3,0.1

Type RM Length L Ch R = 1,110549,1161,1161,1161
BEGIN DESCRIPTION:
Cedar Creek 110549.03
END DESCRIPTION:
XS GIS Cut Line= 3
      1582249.27      6805704.68      1585504.44      6804524.14
      1587448.84      6804124.85
#Sta/Elev= 30
  1534.7 1873.74  1598.8 1872.53  1732.3 1862.54  1919.7 1853.71  2154.0 1850.87
  2264.1 1846.75  2370.5 1848.09  2419.0 1844.16  2628.0 1840.00  3253.4 1831.63
  4370.3 1827.23  4563.9 1823.97  4817.1 1825.48  4891.5 1821.12  4976.7 1821.61
  4987.3 1818.09  4987.5 1815.99  4988.0 1815.49  5007.5 1815.99  5038.7 1822.37
  5098.7 1820.37  5171.4 1823.56  5592.8 1827.58  5735.9 1828.34  5835.0 1826.88
  5937.1 1830.70  6096.0 1838.70  6284.2 1852.27  6544.1 1855.38  6982.3 1854.66
#Mann=5,-1,0
  1534.7    0.05       0  4987.5    0.05       0  5007.5    0.05       0
  5592.8    0.12       0  5735.9    0.05       0
Bank Sta=4987.5,5007.5
Exp/Cntr=0.3,0.1

Type RM Length L Ch R = 1,109388,1153,1153,1153
BEGIN DESCRIPTION:
Cedar Creek 109388.1
END DESCRIPTION:
XS GIS Cut Line= 3
      1582752.70      6806642.20      1585695.41      6805531.09
      1587744.01      6804749.84
#Sta/Elev= 30
  1854.5 1878.15  1967.3 1875.79  2418.3 1854.25  2551.7 1855.78  2583.4 1849.85
  2643.7 1846.64  3380.5 1830.09  3684.8 1827.97  3738.2 1818.49  3770.3 1819.85
  3813.1 1831.21  3855.8 1824.92  3946.9 1823.51  4871.3 1821.46  4939.4 1819.51
  4956.8 1812.15  4972.1 1811.32  4972.6 1810.82  4988.7 1810.82  4992.2 1811.32
  4997.3 1820.30  5034.9 1819.64  5994.9 1822.48  6069.8 1826.42  6202.5 1826.98
  6348.1 1840.66  6451.9 1845.80  6596.9 1845.84  6706.6 1849.90  7192.5 1850.41
#Mann=5,-1,0
  1854.5    0.05       0  4972.1    0.07       0  4988.7    0.12       0
  4992.2    0.05       0  5034.9    0.05       0
Bank Sta=4972.1,4992.2
Exp/Cntr=0.3,0.1

Type RM Length L Ch R = 1,108235,1124,1124,1124
BEGIN DESCRIPTION:
Mapping XS 726ba1b2
END DESCRIPTION:
XS GIS Cut Line= 4
      1583275.06      6807166.89      1584847.98      6806948.14
      1587087.56      6805963.77      1588056.29      6805333.57
#Sta/Elev= 30
  1820.6 1871.00  2067.3 1860.92  2093.1 1857.56  2133.5 1860.26  2163.8 1857.64
  2210.5 1859.86  2244.6 1855.38  2358.9 1850.45  3151.9 1842.91  3770.3 1832.60
  3863.7 1832.97  4082.6 1828.65  4293.5 1815.58  4410.2 1818.51  4745.7 1819.19
  4781.7 1819.85  4825.4 1816.56  4956.5 1818.32  4985.4 1809.05  4985.9 1808.55
  5005.6 1809.05  5008.8 1812.37  5043.9 1817.02  5082.0 1817.87  5136.5 1817.46
  5287.5 1827.46  5393.4 1830.55  5863.9 1834.00  6210.3 1842.38  7010.7 1845.54
#Mann=5,-1,0
  1820.6    0.05       0  4745.7    0.12       0  4985.4    0.07       0
  5005.6    0.12       0  5082.0    0.05       0
Bank Sta=4985.4,5005.6
Exp/Cntr=0.3,0.1

Type RM Length L Ch R = 1,107111,1434,1434,1434
BEGIN DESCRIPTION:
Cedar Creek 107110.57
END DESCRIPTION:
XS GIS Cut Line= 3
      1583246.64      6808454.69      1586215.38      6807061.47
      1588272.68      6806332.30
#Sta/Elev= 30
  1710.0 1869.06  1970.3 1867.93  2448.7 1857.50  2503.5 1861.23  2534.5 1857.83
  2591.9 1858.75  2636.8 1852.77  3376.2 1841.94  3594.3 1834.79  3840.1 1837.40
  4659.7 1830.50  4765.4 1822.60  4872.4 1816.91  4984.6 1815.12  4987.6 1806.28
  4994.8 1806.00  4995.3 1805.50  5015.1 1806.00  5046.0 1815.92  5056.2 1815.69
  5148.9 1815.78  5493.3 1815.57  5549.8 1812.84  5698.9 1816.81  6058.8 1818.07
  6262.1 1821.98  6431.9 1838.32  6516.8 1840.88  6909.3 1843.02  7172.1 1840.58
#Mann=7,-1,0
  1710.0    0.05       0  4765.4    0.12       0  4872.4    0.05       0
  4994.8   0.035       0  5015.1    0.05       0  5056.2    0.12       0
  5148.9    0.05       0
Bank Sta=4994.8,5015.1
Exp/Cntr=0.3,0.1

Type RM Length L Ch R = 1,105677,1198,1198,1198
BEGIN DESCRIPTION:
Mapping XS 5d2bff82
END DESCRIPTION:
XS GIS Cut Line= 4
      1584238.64      6808807.50      1585972.98      6808172.10
      1588045.89      6806984.60      1588451.05      6806496.33
#Sta/Elev= 30
  2079.8 1863.70  2092.4 1861.75  2153.4 1862.86  2209.1 1857.01  2651.0 1845.55
  3660.0 1832.46  4004.8 1830.78  4107.0 1823.19  4159.7 1817.05  4232.3 1815.75
  4521.7 1814.24  4612.0 1813.67  4643.6 1810.14  4680.7 1814.10  4932.1 1813.77
  4977.9 1813.94  4986.5 1804.60  4987.0 1804.10  5006.8 1804.60  5024.0 1813.75
  5144.4 1815.46  5242.9 1814.81  5557.3 1814.17  5653.6 1811.89  5807.7 1820.68
  5916.9 1831.50  5975.9 1840.97  6093.9 1844.18  6320.1 1844.60  6950.3 1839.27
#Mann=9,-1,0
  2079.8    0.05       0  4232.3    0.12       0  4521.7    0.05       0
  4680.7    0.12       0  4932.1    0.05       0  4986.5   0.035       0
  5006.8    0.05       0  5144.4    0.12       0  5242.9    0.05       0
Bank Sta=4986.5,5006.8
Exp/Cntr=0.3,0.1

Type RM Length L Ch R = 1,104479,2006,2006,2006
BEGIN DESCRIPTION:
Cedar Creek 104479.11
END DESCRIPTION:
XS GIS Cut Line= 3
      1585321.70      6809978.58      1587372.50      6808448.62
      1588598.60      6806614.89
#Sta/Elev= 30
  2446.3 1841.84  2562.7 1841.77  2591.7 1844.91  2627.1 1837.70  2949.5 1829.21
  3671.6 1834.38  3713.3 1832.67  3785.4 1812.66  3835.3 1810.80  4234.5 1810.35
  4257.5 1808.33  4625.3 1812.11  4783.3 1812.35  4788.6 1812.40  4941.4 1812.57
  4999.7 1812.22  5000.3 1804.73  5000.8 1804.23  5020.8 1804.73  5036.1 1812.27
  5057.8 1811.70  5074.1 1811.53  5583.1 1810.08  5944.0 1812.76  6081.1 1822.67
  6153.2 1837.00  6219.2 1846.26  6390.4 1847.50  6750.8 1840.36  7210.8 1836.95
#Mann=9,-1,0
  2446.3    0.05       0  4625.3    0.12       0  4783.3    0.05       0
  4788.6    0.12       0  4941.4    0.05       0  5000.3   0.035       0
  5020.8    0.05       0  5057.8    0.12       0  5074.1    0.05       0
#XS Ineff=2,0
    0.00 4647.80 1820.68 5352.20    0.00 1820.68
Permanent Ineff=
       F       F
Bank Sta=5000.3,5020.8
Exp/Cntr=0.3,0.1

Type RM Length L Ch R = 1,102473,920,920,920
BEGIN DESCRIPTION:
Mapping XS d522e485
END DESCRIPTION:
XS GIS Cut Line= 5
      1585400.04      6810385.66      1586488.60      6809557.52
      1587545.89      6809041.89      1588499.02      6808979.39
      1589780.11      6807698.30
#Sta/Elev= 30
  2235.8 1841.17  2473.0 1838.54  2766.1 1840.87  3294.2 1836.15  3564.6 1837.02
  3603.6 1831.23  3632.0 1822.78  3677.1 1813.50  3710.8 1810.54  4161.4 1806.51
  4723.3 1809.60  4999.5 1806.33  4999.6 1800.10  5000.0 1799.60  5016.0 1800.10
  5029.5 1800.99  5039.6 1805.83  5066.6 1808.73  5330.2 1807.29  5374.8 1812.62
  5430.4 1807.27  5450.4 1800.65  5510.6 1800.89  5526.3 1806.97  5560.7 1809.73
  6440.3 1815.49  6511.0 1819.56  6921.1 1821.29  7274.7 1830.13  7546.8 1829.58
#Mann=3,-1,0
  2235.8    0.05       0  4999.6   0.035       0  5016.0    0.05       0
#XS Ineff=2,0
    0.00 4678.30 1819.77 5321.70    0.00 1819.77
Permanent Ineff=
       F       F
Bank Sta=4999.6,5016
Exp/Cntr=0.3,0.1

Type RM Length L Ch R = 1,101553,2116,2116,2116
BEGIN DESCRIPTION:
Cedar Creek 101553.36
END DESCRIPTION:
XS GIS Cut Line= 3
      1585419.40      6810944.27      1588240.55      6809446.89
      1590323.89      6807667.36
#Sta/Elev= 30
  1825.4 1845.43  2884.6 1845.79  2942.6 1843.54  2985.8 1841.95  3141.4 1843.64
  3216.6 1833.31  3238.6 1823.64  3260.5 1819.67  3394.1 1800.62  3552.9 1792.46
  3553.9 1791.96  3593.9 1792.46  3601.0 1797.84  3617.3 1796.86  3705.3 1807.38
  3935.8 1804.22  3957.8 1800.83  3994.1 1803.93  4023.7 1801.33  4474.1 1801.47
  4896.9 1807.48  4962.8 1805.93  5001.2 1799.87  5028.5 1805.42  5149.3 1810.22
  5198.7 1801.37  5262.4 1807.28  6120.9 1814.35  6617.1 1826.06  7759.2 1828.05
#Mann=7,-1,0
  1825.4    0.05       0  2884.6   0.075       0  2942.6    0.05       0
  2985.8   0.075       0  3141.4    0.05       0  3552.9   0.035       0
  3593.9    0.05       0
#XS Ineff=1,-1
 3732.00 6959.40 1812.52
Permanent Ineff=
       F
Bank Sta=3552.9,3593.9
Exp/Cntr=0.3,0.1

Type RM Length L Ch R = 1,99437,1009,1009,1009
BEGIN DESCRIPTION:
Cedar Creek 99436.7
END DESCRIPTION:
XS GIS Cut Line= 3
      1586369.04      6810772.40      1588014.86      6810355.74
      1589848.16      6810251.58
#Sta/Elev= 30
  3311.3 1847.44  3390.0 1847.30  3482.5 1842.66  3595.7 1844.88  3920.5 1843.59
  3961.5 1836.81  4038.3 1817.97  4132.4 1805.19  4183.9 1789.80  4235.4 1788.22
  4236.4 1787.72  4277.0 1788.22  4315.5 1788.68  4418.4 1791.68  4617.5 1796.63
  4658.5 1800.95  4689.2 1808.12  4751.3 1803.35  4940.4 1802.60  4976.3 1793.33
  5019.2 1802.46  5269.6 1805.82  5349.7 1801.24  5379.8 1803.75  5399.8 1800.64
  5469.9 1805.97  5890.6 1803.01  6401.4 1807.92  6661.8 1815.72  6845.3 1817.09
#Mann=7,-1,0
  3311.3    0.05       0  3390.0   0.075       0  3595.7    0.05       0
  4235.4   0.035       0  4277.0    0.05       0  4315.5     0.1       0
  4418.4    0.05       0
Bank Sta=4235.4,4277
Exp/Cntr=0.3,0.1

Type RM Length L Ch R = 1,98428,832,832,832
BEGIN DESCRIPTION:
Cedar Creek 98428.23
END DESCRIPTION:
XS GIS Cut Line= 3
      1586061.72      6811116.16      1587702.36      6810959.91
      1589827.36      6810381.78
#Sta/Elev= 30
  3348.3 1837.34  3379.2 1835.35  3624.8 1840.92  3824.2 1842.64  3904.0 1838.35
  3909.0 1839.33  3964.4 1827.00  4012.0 1819.09  4185.3 1808.92  4295.8 1797.43
  4576.4 1788.44  4577.4 1787.94  4618.0 1788.44  4621.8 1788.48  4721.5 1791.13
  4868.4 1793.69  4908.6 1801.47  4918.7 1801.72  4948.8 1800.28  4968.9 1794.00
  4978.9 1793.52  4995.2 1797.51  5023.8 1800.59  6090.9 1802.81  6190.9 1802.24
  6222.0 1799.97  6314.0 1803.45  6760.9 1806.71  7071.8 1815.61  7198.6 1816.33
#Mann=7,-1,0
  3348.3    0.05       0  3624.8   0.075       0  3824.2    0.05       0
  4576.4   0.035       0  4618.0    0.05       0  4621.8     0.1       0
  4721.5    0.05       0
Bank Sta=4576.4,4618
Exp/Cntr=0.3,0.1

Type RM Length L Ch R = 1,97596,1886,1886,1886
BEGIN DESCRIPTION:
Cedar Creek 97595.94
END DESCRIPTION:
XS GIS Cut Line= 3
      1586332.60      6812220.31      1587994.02      6811683.87
      1589701.17      6810726.20
#Sta/Elev= 30
  3247.2 1849.26  3535.0 1840.24  3575.5 1836.50  3599.1 1828.73  3712.1 1827.23
  3855.4 1815.87  4405.2 1800.84  4474.6 1796.01  4594.8 1797.02  4615.8 1800.41
  4901.5 1800.22  4969.8 1787.78  4970.3 1787.28  4990.6 1787.78  4991.0 1796.85
  4997.4 1797.88  5005.7 1794.68  5035.0 1793.29  5040.8 1795.88  5051.0 1794.17
  5056.7 1797.60  5072.7 1795.28  5121.8 1798.46  5475.8 1800.04  5542.8 1797.76
  5915.9 1800.18  6143.0 1796.52  6224.0 1800.69  6645.0 1803.57  6950.5 1812.52
#Mann=3,-1,0
  3247.2    0.05       0  4969.8   0.035       0  4990.6    0.05       0
#XS Ineff=2,0
    0.00 4747.70 1812.24 5252.30    0.00 1812.24
Permanent Ineff=
       F       F
Bank Sta=4969.8,4990.6
Exp/Cntr=0.3,0.1

Type RM Length L Ch R = 1,95710,1829,1829,1829
BEGIN DESCRIPTION:
Cedar Creek 95710.1
END DESCRIPTION:
XS GIS Cut Line= 3
      1586452.51      6812470.26      1589412.60      6812070.96
      1590089.70      6811489.35
#Sta/Elev= 30
  2018.4 1848.59  2313.5 1843.22  2370.5 1832.22  2448.3 1822.48  2464.9 1818.04
  2626.3 1814.06  2656.6 1808.81  2727.3 1805.94  3045.1 1800.14  3585.0 1795.64
  3642.0 1799.21  3917.9 1799.44  4281.2 1798.71  4382.1 1792.67  4412.4 1796.25
  4493.1 1797.66  4654.6 1795.46  4957.3 1795.85  4986.3 1790.23  4988.4 1786.10
  4988.9 1785.60  5009.3 1786.10  5010.2 1790.48  5016.3 1795.78  5037.1 1794.12
  5059.1 1797.70  5094.2 1798.91  5307.1 1800.56  5555.1 1798.55  5897.9 1805.05
#Mann=3,-1,0
  2018.4    0.05       0  4988.4   0.035       0  5009.3    0.05       0
#XS Ineff=2,0
    0.00 4433.10 1806.25 5566.90    0.00 1806.25
Permanent Ineff=
       F       F
Bank Sta=4988.4,5009.3
Exp/Cntr=0.3,0.1

Type RM Length L Ch R = 1,93881,874,874,874
BEGIN DESCRIPTION:
Cedar Creek 93945.7
END DESCRIPTION:
XS GIS Cut Line= 4
      1586426.46      6812591.79      1588956.05      6812645.62
      1590233.83      6812597.01      1592428.27      6812249.79
#Sta/Elev= 30
  2480.3 1847.70  2668.9 1845.83  2768.9 1840.68  2958.9 1817.79  3149.0 1806.72
  3289.0 1802.33  3579.1 1798.46  3939.2 1798.81  4029.2 1795.39  4199.2 1797.01
  4379.3 1793.32  4509.3 1796.22  4779.4 1795.86  4969.4 1793.33  4989.3 1784.64
  4989.8 1784.14  5010.2 1784.64  5039.4 1794.03  5289.6 1793.74  5469.7 1798.20
  5589.8 1796.60  5850.0 1799.18  5871.8 1798.26  5890.0 1787.56  5945.0 1789.19
  5960.1 1790.22  5970.1 1787.13  6020.1 1795.26  6111.2 1798.85  8510.9 1815.80
#Mann=5,-1,0
  2480.3    0.05       0  4989.3   0.035       0  5010.2    0.05       0
  5945.0    0.12       0  6111.2    0.05       0
#XS Ineff=2,0
    0.00 4580.60 1808.07 5419.40    0.00 1808.07
Permanent Ineff=
       F       F
Bank Sta=4989.3,5010.2
Exp/Cntr=0.3,0.1

Type RM Length L Ch R = 1,93007,350,350,350
BEGIN DESCRIPTION:
Cedar Creek 93007.59
END DESCRIPTION:
XS GIS Cut Line= 3
      1586548.00      6813199.43      1589299.75      6813129.98
      1592636.62      6812789.72
#Sta/Elev= 30
  2242.4 1843.11  2479.5 1837.05  2500.8 1832.80  2609.5 1831.43  2679.5 1821.58
  2779.6 1814.21  2919.6 1813.13  2969.6 1807.51  3129.7 1802.45  3579.8 1797.58
  3879.9 1797.75  4050.0 1795.55  4078.9 1791.69  4140.0 1789.85  4190.0 1794.13
  4810.2 1797.13  4970.3 1791.96  4997.8 1779.91  4998.3 1779.41  5022.7 1779.91
  5040.5 1791.57  5080.7 1793.93  5221.4 1793.51  5372.2 1798.16  5543.1 1794.62
  5960.6 1797.76  6176.8 1799.18  6421.6 1801.28  6474.7 1802.38  8349.2 1814.44
#Mann=7,-1,0
  2242.4    0.05       0  4997.8    0.05       0  5022.7    0.05       0
  5960.6    0.12       0  6176.8    0.05       0  6421.6    0.12       0
  6474.7    0.05       0
#XS Ineff=2,0
    0.00 4653.50 1808.00 5346.50    0.00 1808.00
Permanent Ineff=
       F       F
Bank Sta=4997.8,5022.7
Exp/Cntr=0.3,0.1

Type RM Length L Ch R = 1,92657,1126,1126,1126
BEGIN DESCRIPTION:
Cedar Creek 92656.94
END DESCRIPTION:
XS GIS Cut Line= 3
      1586469.89      6813347.00      1589516.76      6813347.00
      1592355.29      6813208.11
#Sta/Elev= 30
  1965.1 1843.43  2190.2 1842.25  2310.2 1838.91  2330.2 1834.65  2430.2 1834.05
  2530.2 1820.97  2700.2 1817.33  2810.2 1809.23  3010.2 1803.42  3430.2 1798.26
  3640.2 1798.91  4010.2 1795.65  4130.2 1792.06  4330.2 1797.47  4640.2 1795.85
  4800.2 1792.03  4950.2 1791.92  4960.2 1791.39  4987.7 1782.99  4988.2 1782.49
  5012.6 1782.99  5020.2 1791.97  5080.3 1789.82  5200.4 1795.66  5768.4 1795.19
  5901.3 1792.54  6091.6 1796.82  6371.8 1801.83  6632.1 1801.86  7853.9 1811.57
#Mann=5,-1,0
  1965.1    0.05       0  4987.7    0.05       0  5012.6    0.05       0
  5768.4    0.12       0  6091.6    0.05       0
#XS Ineff=2,0
    0.00 4452.60 1806.37 5547.40    0.00 1806.37
Permanent Ineff=
       F       F
Bank Sta=4987.7,5012.6
Exp/Cntr=0.3,0.1

Type RM Length L Ch R = 1,91531,910,910,910
BEGIN DESCRIPTION:
Cedar Creek 91531.26
END DESCRIPTION:
XS GIS Cut Line= 3
      1586504.64      6814267.14      1589212.94      6814232.41
      1592216.45      6814006.72
#Sta/Elev= 30
  2299.9 1837.03  2618.9 1833.68  2640.3 1832.55  2650.3 1828.69  2760.3 1827.60
  2820.3 1820.98  2890.3 1819.42  2920.3 1816.13  3300.3 1806.54  3810.4 1800.04
  4150.4 1791.31  4184.0 1790.12  4210.4 1785.91  4290.4 1792.46  4920.5 1791.85
  4970.5 1790.27  4990.2 1780.17  4990.6 1779.67  5010.2 1780.17  5012.0 1783.70
  5020.5 1788.77  5030.5 1789.86  5194.4 1790.70  5213.0 1790.79  5398.8 1794.72
  5872.9 1790.40  6103.6 1792.32  6153.7 1789.13  6635.1 1796.70  8020.4 1810.63
#Mann=5,-1,0
  2299.9    0.05       0  4990.2    0.05       0  5010.2    0.05       0
  5194.4    0.12       0  5213.0    0.05       0
#XS Ineff=2,0
    0.00 4588.10 1805.36 5411.90    0.00 1805.36
Permanent Ineff=
       F       F
Bank Sta=4990.2,5010.2
Exp/Cntr=0.3,0.1

Type RM Length L Ch R = 1,90621,561,561,561
BEGIN DESCRIPTION:
Cedar Creek 90621.36
END DESCRIPTION:
XS GIS Cut Line= 3
      1586669.50      6814787.97      1589065.37      6815013.66
      1592225.10      6814978.94
#Sta/Elev= 30
  2604.6 1826.67  2977.4 1811.10  3293.1 1801.99  4047.9 1788.74  4357.8 1790.03
  4528.6 1786.66  4598.9 1790.25  4920.3 1790.63  4950.4 1789.80  4982.3 1779.89
  4982.7 1779.39  5002.2 1779.89  5008.4 1783.95  5020.7 1786.32  5050.7 1788.83
  5650.7 1786.78  5930.8 1790.76  6020.8 1788.71  6050.8 1790.19  6200.8 1785.50
  6300.8 1788.66  6520.8 1788.98  6540.8 1797.20  6570.8 1792.37  6610.8 1780.94
  6660.8 1780.63  6740.8 1782.02  6810.8 1797.19  6850.8 1791.54  8171.0 1806.84
#Mann=3,-1,0
  2604.6    0.05       0  4982.3    0.05       0  5002.2    0.05       0
#XS Ineff=2,0
       0                 5781.30    0.00 1801.44
Permanent Ineff=
       F       F
Bank Sta=4982.3,5002.2
Exp/Cntr=0.3,0.1
