HEC-RAS study Cedar Creek 2.prj: Cedar Creek 2 Base Level Engineering

--- Cedar Creek 2.g01 (geometry) --- (continued)

Type RM Length L Ch R = 1 ,24589   ,222,222,222
BEGIN DESCRIPTION:
564
END DESCRIPTION:
XS GIS Cut Line= 3
      1509124.25       6790935.3      1508655.49      6790956.14
      1507968.95      6791109.57
#Sta/Elev= 30
  4530.8 2277.99  4560.1 2278.26  4680.2 2274.78  4699.7 2275.15  4720.2    2273
  4760.3 2262.09  4780.3 2258.19  4820.3 2255.24  4869.9 2254.43  4932.4 2253.29
  4950.5 2249.67  4960.5 2244.73  4970.5 2243.94    4976 2242.19  4976.5 2241.69
    4985 2242.19  4990.5 2242.93  4997.8 2245.92    5021 2248.46  5101.7 2248.71
  5125.9 2247.93  5133.7 2251.31  5154.2 2265.98  5164.2 2274.43  5169.3 2274.48
    5185 2297.48  5195.2 2302.25  5328.4  2306.4  5523.1 2304.47  5703.5 2308.58
#Mann= 5 ,-1 , 0
  4530.8     .16       0  4869.9     .07       0    4976     .07       0
    4985     .07       0  5101.7     .16       0
Bank Sta=4976,4985
XS Rating Curve= 0 ,0
Exp/Cntr=0.3,0.1

Type RM Length L Ch R = 1 ,24367   ,134,134,134
BEGIN DESCRIPTION:
565
END DESCRIPTION:
XS GIS Cut Line= 3
      1509119.05      6790854.58      1508647.68      6790732.18
      1508048.03       6790719.2
#Sta/Elev= 30
    4521 2276.82  4597.5 2275.66  4659.5 2276.26  4731.8  2275.5    4767 2273.88
  4802.4 2259.05  4807.6 2258.67  4814.5 2255.57  4824.8 2253.52  4837.1 2252.38
  4924.1 2250.65  4938.5 2245.99  4990.1 2243.35  4995.5 2239.95    4996 2239.45
  5004.5 2239.95  5009.9 2240.54  5011.8 2240.54  5020.7 2244.69  5030.7 2246.38
  5080.7 2248.15  5140.7 2252.12  5150.7 2253.65  5170.7 2260.78  5230.7 2287.51
  5260.7 2290.43  5300.8 2297.59  5440.8 2304.55  5480.8 2307.26  5607.8 2311.39
#Mann= 5 ,-1 , 0
    4521     .16       0  4837.1     .07       0  4995.5     .07       0
  5004.5     .07       0  5009.9     .16       0
Bank Sta=4995.5,5004.5
XS Rating Curve= 0 ,0
Exp/Cntr=0.3,0.1

Type RM Length L Ch R = 1 ,24233   ,234,234,234
BEGIN DESCRIPTION:
563
END DESCRIPTION:
XS GIS Cut Line= 3
      1509095.64      6790768.65      1508652.89      6790599.37
      1508079.95      6790607.18
#Sta/Elev= 30
  4529.3 2274.56  4669.2  2274.8  4701.3 2273.39  4721.6 2270.23  4776.2 2254.59
  4794.7 2252.02  4872.6 2250.74    4894 2242.83  4909.6 2242.19  4958.2 2243.84
  4973.1 2239.78    4975  2239.3  4975.5  2238.8  4984.2  2239.3  5021.2 2246.07
  5091.2 2247.97  5101.2 2250.41  5111.2 2255.71  5121.2 2264.06  5131.2  2269.4
  5141.2 2271.99  5151.2 2271.51  5171.2 2266.84  5181.2 2267.57  5201.2 2273.89
  5211.2  2282.2  5221.2 2287.74    5268 2290.08  5301.2 2298.14  5576.3 2311.12
#Mann= 5 ,-1 , 0
  4529.3     .16       0  4721.6     .07       0  4973.1     .16       0
    4975     .07       0  4984.2     .16       0
Bank Sta=4975,4984.2
XS Rating Curve= 0 ,0
Exp/Cntr=0.3,0.1

Type RM Length L Ch R = 1 ,23999   ,156,156,156
BEGIN DESCRIPTION:
562
END DESCRIPTION:
XS GIS Cut Line= 3
      1509158.11      6790779.07      1508832.57      6790461.35
      1508226.35       6790242.8
#Sta/Elev= 30
  4544.4 2273.85  4639.3 2273.63  4722.7 2268.68  4745.3 2266.77  4752.4 2268.51
  4759.4 2266.68  4766.6 2267.86  4773.6 2265.41  4780.7 2266.26  4787.7 2263.85
  4844.3 2254.73  4929.2 2246.11  4950.5 2239.02  4964.6    2238  4981.2 2234.01
  4981.7 2233.51  4990.4 2234.01  5028.9 2241.77  5071.1 2244.74    5168 2244.54
  5197.1  2245.5  5209.3 2248.69  5219.9 2253.13  5251.8 2272.16  5258.5 2278.18
  5273.1 2283.86  5375.9 2288.88  5381.2 2287.72  5462.6 2297.02  5643.7 2306.31
#Mann= 5 ,-1 , 0
  4544.4     .16       0  4722.7     .07       0  4981.2     .07       0
  4990.4     .07       0    5168     .16       0
Bank Sta=4981.2,4990.4
XS Rating Curve= 0 ,0
Exp/Cntr=0.3,0.1

Type RM Length L Ch R = 1 ,23843   ,226,226,226
BEGIN DESCRIPTION:
561
END DESCRIPTION:
XS GIS Cut Line= 3
      1509184.15      6790724.38      1508934.14      6790362.39
      1508415.88      6790117.58
#Sta/Elev= 30
  4558.4 2268.36  4583.8 2272.54  4649.4 2273.05  4683.2  2271.5  4691.3 2271.64
  4706.2 2268.15  4712.3 2269.05  4721.1 2266.59  4727.1 2267.99  4735.9 2265.58
    4742 2267.19  4756.9 2261.89    4763 2262.85  4792.7 2255.37  4857.8 2252.17
  4965.8 2243.97  4993.4 2232.57  4993.9 2232.07  5002.6 2232.57  5017.1 2239.06
  5062.7 2239.28  5113.7    2243  5174.2 2242.71  5210.3  2242.9  5227.6 2249.94
  5240.7 2258.25  5262.8 2269.23  5278.6 2271.48  5406.6 2272.96  5571.5  2286.5
#Mann= 5 ,-1 , 0
  4558.4     .16       0  4683.2     .07       0  4993.4     .07       0
  5002.6     .07       0  5174.2     .16       0
Bank Sta=4993.4,5002.6
XS Rating Curve= 0 ,0
Exp/Cntr=0.3,0.1

Type RM Length L Ch R = 1 ,23617   ,235,235,235
BEGIN DESCRIPTION:
560
END DESCRIPTION:
XS GIS Cut Line= 3
       1509449.8      6790206.14      1508996.64      6790161.87
      1508504.42      6790086.34
#Sta/Elev= 30
  4553.6 2294.24  4558.5 2294.24  4584.7 2288.39  4589.7 2289.39  4628.8 2283.17
  4658.9 2276.85    4679  2269.9  4686.4 2264.94  4699.1 2259.65  4729.2 2252.85
  4799.6 2246.73  4965.7 2242.91  4970.4 2242.72  4990.5 2233.92  4996.5 2232.59
    4997 2232.09  5006.3 2232.59  5007.2 2234.08  5012.3 2234.08  5020.7  2236.7
  5091.5 2239.45  5112.6 2239.07  5142.1 2238.53  5152.2 2240.79  5198.5 2261.09
  5203.6  2264.9    5223 2263.98  5243.3 2267.51    5304  2271.2  5506.9 2276.41
#Mann= 5 ,-1 , 0
  4553.6     .16       0  4965.7     .07       0  4996.5     .07       0
  5006.3     .07       0  5112.6     .16       0
Bank Sta=4996.5,5006.3
XS Rating Curve= 0 ,0
Exp/Cntr=0.3,0.1

Type RM Length L Ch R = 1 ,23382   ,131,131,131
BEGIN DESCRIPTION:
559
END DESCRIPTION:
XS GIS Cut Line= 3
       1509488.8      6789956.14      1509043.51      6789940.51
      1508475.78      6790016.04
#Sta/Elev= 30
  4557.1 2302.02  4590.9 2298.66  4620.9 2287.89  4646.3 2281.69  4651.3 2283.45
    4661 2282.55    4691 2276.16    4741 2271.83    4751 2269.67    4761 2265.69
    4781 2254.04  4801.1  2245.3  4821.1 2241.97  4871.1 2239.33  4981.2 2238.41
  4991.2 2233.35  4994.5 2227.79    4995 2227.29  5004.3 2227.79  5011.3 2229.01
  5018.9 2235.28    5024 2233.58  5031.4 2235.61  5098.4 2234.57  5112.1 2235.58
  5142.4 2252.52  5152.5 2256.07  5182.8  2264.1  5202.9 2266.26  5575.4 2276.28
#Mann= 4 ,-1 , 0
  4557.1     .07       0  4994.5     .07       0  5004.3     .07       0
  5098.4     .16       0
Bank Sta=4994.5,5004.3
XS Rating Curve= 0 ,0
Exp/Cntr=0.3,0.1

Type RM Length L Ch R = 1 ,23251   ,285,285,285
BEGIN DESCRIPTION:
557
END DESCRIPTION:
XS GIS Cut Line= 3
      1509470.57      6789864.99      1508999.24      6789823.33
      1508413.62      6789943.05
#Sta/Elev= 30
    4533 2295.12  4538.6 2291.98  4554.6 2288.51  4628.9 2282.31  4655.3 2276.22
  4666.6 2272.83  4671.6 2267.89  4729.6 2247.68  4759.4  2240.8  4809.6 2237.72
  4950.2 2237.23  4970.3 2235.94  4980.3 2234.71  5000.4  2224.5  5000.9 2222.89
  5001.4 2222.39  5010.7 2222.89  5020.7 2229.63  5030.9 2233.25    5087 2233.83
  5122.8 2232.66    5133 2234.36  5143.2 2238.77  5163.6 2257.49  5201.8 2266.61
  5257.4 2268.05  5347.3 2266.99  5510.6 2274.38  5571.9 2275.63  5603.9 2278.54
#Mann= 6 ,-1 , 0
    4533     .07       0  4655.3     .16       0  4729.6     .07       0
  5000.9     .07       0  5010.7     .07       0    5087     .16       0
Bank Sta=5000.9,5010.7
XS Rating Curve= 0 ,0
Exp/Cntr=0.3,0.1

Type RM Length L Ch R = 1 ,22966   ,149,149,149
BEGIN DESCRIPTION:
558
END DESCRIPTION:
XS GIS Cut Line= 3
      1509423.73      6789628.01      1509150.28       6789620.2
      1508494.08      6789651.45
#Sta/Elev= 30
  4730.6 2300.51  4779.3 2296.19  4799.4 2288.59  4809.4  2279.8  4849.4 2251.39
  4869.4 2240.18  4905.3 2234.45  4936.4 2234.83  4959.4    2235  4979.4 2227.21
  4984.5 2226.28    4985 2225.78  4994.4 2226.28  4999.3 2229.14  5004.2 2229.14
  5009.4 2230.88  5039.5 2232.41  5058.7 2234.84  5063.8 2232.89  5069.5 2235.34
  5079.5 2236.48  5329.8  2236.1  5439.9 2240.74    5460 2245.47  5479.2  2251.9
    5490  2258.3    5500 2260.65    5530 2265.06  5593.1 2267.25  5661.1 2269.34
#Mann= 5 ,-1 , 0
  4730.6     .16       0  4936.4     .07       0  4984.5     .07       0
  4994.4     .07       0  5593.1     .16       0
Bank Sta=4984.5,4994.4
XS Rating Curve= 0 ,0
Exp/Cntr=0.3,0.1

Type RM Length L Ch R = 1 ,22817   ,383,383,383
BEGIN DESCRIPTION:
556
END DESCRIPTION:
XS GIS Cut Line= 3
       1509488.8      6789489.99      1509204.97      6789487.39
      1508540.88      6789544.68
#Sta/Elev= 30
  4716.6 2308.14  4830.4 2301.71  4847.2 2291.89  4880.4 2271.97  4900.4 2257.42
  4920.4 2246.15  4940.4 2237.97  4950.4  2236.5  4970.4 2228.63  4985.5 2225.45
    4986 2224.95  4995.4 2225.45  5002.9 2226.13  5010.4 2229.77  5028.1 2230.38
  5040.6 2231.12  5050.6 2233.33  5070.7 2234.54  5191.1 2235.69  5297.5  2234.4
  5466.8 2235.36  5502.3 2237.31  5529.2 2242.47  5534.2 2241.75  5552.5 2248.14
  5562.5 2249.87  5602.6 2261.48  5622.7 2263.72  5656.2 2264.83    5667 2265.09
#Mann= 7 ,-1 , 0
  4716.6     .07       0  4847.2     .16       0  4985.5     .07       0
  4995.4     .16       0  5028.1     .07       0  5466.8     .16       0
  5656.2     .07       0
Bank Sta=4985.5,4995.4
XS Rating Curve= 0 ,0
Exp/Cntr=0.3,0.1

Type RM Length L Ch R = 1 ,22434   ,263,263,263
BEGIN DESCRIPTION:
555
END DESCRIPTION:
XS GIS Cut Line= 3
      1509405.46      6789159.26      1509001.85       6789180.1
      1508528.96      6789421.74
#Sta/Elev= 30
    4592 2302.62  4742.7 2302.15  4809.4 2300.05  4822.8 2298.83  4832.8 2294.95
  4842.8 2285.75  4852.8 2273.91  4858.1 2264.98  4863.1  2261.6  4912.9 2235.89
  4922.9 2231.34  4934.7 2228.31    4983 2226.18  4995.4 2222.95  4995.9 2222.45
  5005.3 2222.95  5037.5 2228.34  5111.5 2226.34  5161.5 2229.79  5289.2 2231.97
  5340.8 2235.26  5355.9 2236.66  5372.5 2242.87  5378.1 2242.74  5394.7 2251.31
  5400.3  2250.8  5416.9 2258.41  5422.5 2258.24  5430.6 2260.54  5527.2 2264.13
#Mann= 6 ,-1 , 0
    4592     .07       0  4809.4     .16       0  4934.7     .07       0
  4995.4     .07       0  5005.3     .07       0  5340.8     .16       0
Bank Sta=4995.4,5005.3
XS Rating Curve= 0 ,0
Exp/Cntr=0.3,0.1

Type RM Length L Ch R = 1 ,22171   ,162,162,162
BEGIN DESCRIPTION:
554
END DESCRIPTION:
XS GIS Cut Line= 3
      1509356.02      6788966.55      1508796.12      6789021.24
      1508512.23      6789341.59
#Sta/Elev= 30
  4446.6 2302.57    4518 2298.17    4546 2289.87  4588.3 2275.21  4608.4 2266.93
  4619.6 2260.72  4648.6 2251.59  4716.3 2244.04  4721.3 2245.49    4739 2244.58
  4836.1 2234.28  4909.8 2229.05    4940 2224.55  5014.9  2225.5  5029.2  2224.6
  5043.4  2222.3  5045.1 2220.53  5045.6 2220.03  5055.1 2220.53  5078.5 2227.17
  5099.4 2227.96  5142.1 2233.87  5168.2 2235.06  5198.9 2235.84  5227.4 2239.52
  5241.6 2242.19  5276.7 2254.92  5298.5 2259.09  5319.4 2260.69  5437.2 2262.65
#Mann= 6 ,-1 , 0
  4446.6     .07       0    4546     .16       0  4836.1     .07       0
  5045.1     .07       0  5055.1     .07       0  5168.2     .16       0
Bank Sta=5045.1,5055.1
XS Rating Curve= 0 ,0
Exp/Cntr=0.3,0.1

Type RM Length L Ch R = 1 ,22009   ,125,125,125
BEGIN DESCRIPTION:
553
END DESCRIPTION:
XS GIS Cut Line= 3
      1509296.09      6788927.49      1508759.66      6788872.81
       1508090.4      6788961.35
#Sta/Elev= 30
  4456.4 2300.71  4517.8 2298.38  4570.6 2285.15  4588.2 2278.45  4596.2  2272.7
  4601.3  2275.5  4608.3 2270.82  4648.5 2255.61  4695.8 2243.66  4728.9 2240.04
  4795.4  2232.3  4989.4 2226.72  5001.2 2222.29  5005.4 2218.52  5005.9 2218.02
  5015.4 2218.52  5030.6 2223.21  5131.4 2224.34  5141.5 2219.16  5171.8  2225.5
  5272.7 2228.11    5305 2238.53  5353.4 2239.94  5373.4 2244.28  5378.5 2241.22
    5424 2254.86  5451.9 2260.05  5456.9  2258.9  5608.8 2264.48  5670.7 2270.08
#Mann= 5 ,-1 , 0
  4456.4     .07       0  4570.6     .16       0  4728.9     .07       0
  5005.4     .07       0  5015.4     .07       0
Bank Sta=5005.4,5015.4
XS Rating Curve= 0 ,0
Exp/Cntr=0.3,0.1

Type RM Length L Ch R = 1 ,21884   ,317,317,317
BEGIN DESCRIPTION:
551
END DESCRIPTION:
XS GIS Cut Line= 3
      1509288.28       6788810.3      1508707.57      6788763.43
      1508061.72      6788922.29
#Sta/Elev= 30
  4414.6 2299.03  4498.1 2298.09  4538.3 2294.31  4578.4 2285.75  4626.6 2257.42
  4631.6 2258.62  4635.9 2255.44  4678.7 2239.93  4734.9 2231.86  4819.2  2227.7
  4959.6 2226.96  4989.7 2219.85    4991 2216.87  4991.5 2216.37    5001 2216.87
  5036.6 2222.23  5071.9 2221.82  5102.8 2217.83  5113.1 2221.14  5136.1 2222.34
  5182.3 2222.82  5238.7 2225.18  5290.9 2226.27  5319.1 2241.23  5339.7 2255.79
    5350 2259.06  5368.8  2257.3  5551.3 2265.12  5649.2 2274.99  5662.3 2276.66
#Mann= 10 ,-1 , 0
  4414.6     .07       0  4635.9     .16       0  4734.9     .07       0
    4991     .07       0    5001     .07       0  5136.1     .16       0
  5182.3     .07       0  5238.7     .16       0  5551.3     .07       0
  5649.2     .16       0
Bank Sta=4991,5001
XS Rating Curve= 0 ,0
Exp/Cntr=0.3,0.1

Type RM Length L Ch R = 1 ,21567   ,248,248,248
BEGIN DESCRIPTION:
552
END DESCRIPTION:
XS GIS Cut Line= 3
      1509288.27      6788786.86      1508621.64      6788588.95
      1507941.95      6788747.81
#Sta/Elev= 30
  4125.6  2297.9  4169.9 2296.75  4175.1 2294.76    4202 2293.86  4213.6  2290.8
  4295.9 2284.37  4306.3 2281.35  4313.2 2275.54  4353.6 2253.49  4400.2 2237.24
    4456 2231.11  4556.1 2225.92  4666.2  2225.4  4723.6 2229.75  4804.3 2231.42
  4920.8 2224.74  4968.5  2220.9  4986.5 2214.87    4987 2214.37  4997.8 2214.87
  5022.9 2218.89  5115.4 2219.11  5148.8 2228.57  5191.3 2245.61  5197.5  2250.4
  5218.1 2259.95  5233.9 2265.13    5324  2268.9    5409 2281.03    5519  2291.5
#Mann= 6 ,-1 , 0
  4125.6     .07       0  4353.6     .16       0    4456     .07       0
  4920.8     .16       0  4986.5     .07       0  4997.8     .16       0
Bank Sta=4986.5,4997.8
XS Rating Curve= 0 ,0
Exp/Cntr=0.3,0.1

Type RM Length L Ch R = 1 ,21319   ,322,322,322
BEGIN DESCRIPTION:
550
END DESCRIPTION:
XS GIS Cut Line= 3
       1509251.8      6788750.39      1508379.45      6788448.33
      1507929.48       6788388.5
#Sta/Elev= 30
  4002.3 2290.27  4125.9 2282.93  4136.5 2279.89  4175.6 2254.78    4194 2247.12
  4212.1 2241.16  4237.9 2235.92  4297.7 2230.61  4432.8 2224.91  4518.3 2225.37
  4559.8 2228.87    4655 2230.47    4700 2229.17  4771.4 2221.16  4898.4 2221.19
  4920.1  2218.8  4960.2 2218.75    5005 2213.57  5005.5 2213.07  5016.3 2213.57
  5030.8 2225.73  5038.8 2229.89  5043.9 2229.78  5071.2 2239.98  5111.5 2249.44
  5141.8 2260.42  5182.2 2269.83  5212.4 2281.63  5323.4 2298.58  5379.4 2303.08
#Mann= 6 ,-1 , 0
  4002.3     .07       0    4194     .16       0  4297.7     .07       0
  4920.1     .16       0    5005     .07       0  5016.3     .16       0
Bank Sta=5005,5016.3
XS Rating Curve= 0 ,0
Exp/Cntr=0.3,0.1

Type RM Length L Ch R = 1 ,20997   ,230,230,230
BEGIN DESCRIPTION:
549
END DESCRIPTION:
XS GIS Cut Line= 3
      1509283.12      6788547.29      1508486.22      6788213.95
      1508072.15       6787997.8
#Sta/Elev= 30
  4131.6  2286.5  4142.9 2285.66  4227.1 2268.69  4244.9 2266.85  4321.7 2247.67
  4345.5 2244.32  4350.9 2246.99  4374.7 2239.06  4380.1 2241.43  4422.2 2230.05
  4466.3  2226.4  4846.4 2217.28  4970.8  2217.7  4985.9 2216.79  4994.3 2211.11
  4994.8 2210.61  5005.6 2211.11  5030.6 2211.25  5044.1 2215.51  5060.6 2215.25
  5082.6 2220.28  5146.1  2225.7    5171 2227.85  5193.1  2233.5  5237.2 2249.07
  5267.5 2262.61  5312.6 2273.25    5342 2283.91  5414.2 2296.19  5462.5 2300.65
#Mann= 6 ,-1 , 0
  4131.6     .07       0  4142.9     .16       0  4466.3     .07       0
  4994.3     .07       0  5005.6     .07       0  5146.1     .16       0
Bank Sta=4994.3,5005.6
XS Rating Curve= 0 ,0
Exp/Cntr=0.3,0.1

Type RM Length L Ch R = 1 ,20767   ,332,332,332
BEGIN DESCRIPTION:
548
END DESCRIPTION:
XS GIS Cut Line= 4
       1509332.6      6788476.99      1508762.28      6788140.05
      1508613.82      6788031.66      1508226.53      6787792.52
#Sta/Elev= 30
  4152.2 2291.18  4218.5 2278.22  4232.8 2274.89  4323.6 2259.48  4444.6 2253.45
  4585.8 2250.62  4660.5 2252.59  4705.8  2247.7  4776.6 2231.41  4799.8 2229.92
  4842.9 2212.53    4985 2213.87  4993.5 2213.14  4997.3 2209.19  5009.1 2208.53
  5009.6 2208.03  5020.5 2208.53  5020.7  2210.5  5044.1 2216.47    5094 2215.54
  5169.5 2218.84  5246.5 2228.59  5261.9 2237.23  5267.8 2237.03  5277.3 2241.53
  5283.2  2240.6  5298.6 2250.41    5314 2256.67  5384.9 2281.94  5453.6 2287.33
#Mann= 8 ,-1 , 0
  4152.2     .07       0  4218.5     .16       0  4232.8     .07       0
  4444.6     .16       0  4585.8     .07       0  5009.1     .07       0
  5020.5     .07       0  5169.5     .16       0
Bank Sta=5009.1,5020.5
XS Rating Curve= 0 ,0
Exp/Cntr=0.3,0.1

Type RM Length L Ch R = 1 ,20435   ,408,408,408
BEGIN DESCRIPTION:
544
END DESCRIPTION:
XS GIS Cut Line= 3
      1509363.81      6788385.81      1508871.64      6788023.85
      1508314.31      6787739.98
#Sta/Elev= 30
  4387.6 2284.29  4421.6 2279.78  4492.6  2264.7  4535.1 2259.62  4613.8 2254.04
  4665.5 2253.18    4718 2252.21  4799.7 2248.92  4857.8 2237.29  4914.6 2230.87
  4920.8 2225.52  4929.3 2222.99  4935.5 2216.19  4943.9  2213.1  4950.1 2208.08
  4959.1 2206.14  4959.6 2205.64  4970.5 2206.14    4971 2209.71  4985.6 2211.75
  5111.6 2211.49    5390 2217.16  5445.2 2221.16  5499.8 2230.37  5522.2 2238.11
  5556.4 2255.14  5567.1 2258.25  5589.6 2270.99  5595.2 2275.85    5624 2281.51
#Mann= 6 ,-1 , 0
  4387.6     .07       0  4665.5     .16       0    4718     .07       0
  4959.1     .07       0  4970.5     .07       0    5390     .16       0
Bank Sta=4959.1,4970.5
XS Rating Curve= 0 ,0
Exp/Cntr=0.3,0.1

Type RM Length L Ch R = 1 ,20027   ,221,221,221
BEGIN DESCRIPTION:
545
END DESCRIPTION:
XS GIS Cut Line= 3
      1509400.25      6788331.11      1508717.99      6787729.58
      1508460.79      6787472.38
#Sta/Elev= 30
  4089.6  2276.3  4116.8 2274.94  4137.7 2267.63  4258.2 2253.33  4449.8 2242.41
  4484.9 2241.41  4492.4  2244.2  4541.8    2237    4648 2230.43  4676.5 2223.17
  4690.7 2213.57  4704.9  2211.9  4776.1 2210.36    4797 2214.65  4825.4  2214.8
  4853.9  2204.7  4860.5 2207.69  4868.1 2204.92  4874.8 2209.27  4909.9 2209.22
  4966.8 2208.23  4982.9 2202.83  4983.4 2202.33  4994.3 2202.83  5016.5 2211.78
  5030.7 2213.15  5214.5 2219.03  5292.3  2259.4  5320.6 2261.78  5362.9 2259.22
#Mann= 3 ,-1 , 0
  4089.6     .07       0  4982.9     .07       0  4994.3     .07       0
Bank Sta=4982.9,4994.3
XS Rating Curve= 0 ,0
Exp/Cntr=0.3,0.1

Type RM Length L Ch R = 1 ,19806   ,213,213,213
BEGIN DESCRIPTION:
547
END DESCRIPTION:
XS GIS Cut Line= 4
      1509400.27      6788279.04      1509009.66      6787898.85
      1508832.57      6787549.89      1508465.39      6787409.27
#Sta/Elev= 30
    3980 2263.78  4062.2 2262.38  4090.5 2261.12  4097.7 2258.61  4104.7 2260.27
  4140.1 2256.15  4295.5 2247.34  4352.1 2238.67  4678.2 2218.63  4895.2 2212.52
  4924.5 2209.03  4956.6  2209.9  4962.8 2206.55  4978.1 2206.31  4981.8 2201.51
  4982.3 2201.01  4993.2 2201.51  5017.5 2209.23  5031.6 2211.34  5072.3 2213.04
  5107.7 2225.22    5127 2228.62  5138.7 2235.33  5157.1 2240.46  5162.4 2244.57
  5181.5 2251.05  5192.4 2257.89  5202.9 2260.46  5266.5 2260.32  5309.6 2254.69
#Mann= 3 ,-1 , 0
    3980     .07       0  4981.8     .07       0  4993.2     .07       0
Bank Sta=4981.8,4993.2
XS Rating Curve= 0 ,0
Exp/Cntr=0.3,0.1

Type RM Length L Ch R = 1 ,19593   ,239,239,239
BEGIN DESCRIPTION:
546
END DESCRIPTION:
XS GIS Cut Line= 4
       1509408.1      6788245.21      1509103.41      6787937.91
      1508777.89      6787312.91      1508723.27      6786782.35
#Sta/Elev= 30
  3863.7 2268.31  3920.5  2265.7  3927.6    2268  3948.8 2264.63    3970  2265.7
  4033.6 2257.01  4146.8 2246.89  4189.2 2245.78  4231.6 2237.37  4330.6 2230.27
  4612.3 2215.16  4984.1 2205.04  4993.2 2204.11  4995.4 2200.63  4995.9 2200.13
  5006.8 2200.63  5026.2 2204.26  5046.3 2211.57  5074.8 2211.75  5079.8 2216.41
  5156.9 2213.42  5178.9 2216.06  5217.2 2209.68  5247.3 2210.63    5278    2216
    5367 2239.14  5438.3 2247.91  5466.2 2256.88    5497 2258.08  5534.5 2259.09
#Mann= 5 ,-1 , 0
  3863.7     .07       0  4995.4     .07       0  5006.8     .07       0
  5466.2     .16       0    5497     .07       0
Bank Sta=4995.4,5006.8
XS Rating Curve= 0 ,0
Exp/Cntr=0.3,0.1

Type RM Length L Ch R = 1 ,19354   ,241,241,241
BEGIN DESCRIPTION:
543
END DESCRIPTION:
XS GIS Cut Line= 3
      1509345.59      6787958.73      1508967.99      6787187.91
       1508895.2      6786712.19
#Sta/Elev= 30
  4141.8 2252.08  4179.4 2249.73  4196.3 2251.01  4201.9 2249.55  4218.8 2249.68
  4276.2 2240.89  4449.4  2222.3  4567.5 2213.78  4652.7 2211.14  4844.1 2206.41
  4882.5 2206.61    4922  2208.8    4950 2208.34  4972.5 2204.47  4988.9 2198.09
  4991.9 2194.37  4992.4 2193.87  5003.9 2194.37  5020.3 2201.86  5070.9 2207.68
  5101.2 2218.06  5122.8 2217.34  5141.7 2220.78  5181.1 2224.48  5270.1 2227.25
  5293.8 2227.81  5354.1  2237.8  5381.5 2240.63  5394.6 2245.85  5481.4 2247.74
#Mann= 6 ,-1 , 0
  4141.8    .035       0  4652.7     .07       0  4991.9     .07       0
  5003.9     .07       0  5270.1     .16       0  5293.8     .07       0
Bank Sta=4991.9,5003.9
XS Rating Curve= 0 ,0
Exp/Cntr=0.3,0.1

Type RM Length L Ch R = 1 ,19113   ,355,355,355
BEGIN DESCRIPTION:
542
END DESCRIPTION:
XS GIS Cut Line= 3
      1509418.51      6787784.25      1509178.93      6787099.37
      1508929.49      6786704.42
#Sta/Elev= 30
  4261.7 2252.96    4410 2249.58  4435.7 2245.58    4441 2246.66  4466.7 2235.44
    4472 2235.76  4497.8 2224.86    4613 2215.38  4692.1 2207.26  4777.1  2206.8
  4808.6  2204.1  4864.6 2205.46  4882.8 2205.13  4890.6 2201.84    4991 2201.75
  5005.3  2200.4  5006.5 2197.44    5007 2196.94  5018.5 2197.44  5041.8 2201.05
  5057.1 2213.23    5063 2213.17  5071.7 2217.53  5124.5 2218.86  5267.5 2225.64
  5278.3 2227.03  5339.4 2234.11  5381.8 2236.69    5403 2245.48  5454.4 2247.33
#Mann= 8 ,-1 , 0
  4261.7     .16       0    4613     .07       0  4864.6     .16       0
  5006.5     .07       0  5018.5     .16       0  5124.5     .07       0
  5267.5     .16       0  5278.3     .07       0
Bank Sta=5006.5,5018.5
XS Rating Curve= 0 ,0
Exp/Cntr=0.3,0.1

Type RM Length L Ch R = 1 ,18758   ,189,189,189
BEGIN DESCRIPTION:
541
END DESCRIPTION:
XS GIS Cut Line= 3
      1509637.28      6787620.24      1509457.57      6787091.56
       1508924.2      6786672.66
#Sta/Elev= 30
  4543.9 2261.78  4603.1 2253.77  4663.2  2251.6  4721.2  2242.7  4757.9 2245.94
  4768.1  2244.9  4778.6 2242.45    4784 2237.48  4789.2 2236.49  4810.1 2223.38
  4815.3 2223.33  4820.9 2217.21  4841.4 2207.94  4863.1 2204.55  4940.9 2203.08
  4972.2 2198.46  4983.8 2192.95  4984.3 2192.45  4995.9 2192.95  4998.3 2196.07
    5011 2200.34    5035 2199.78  5074.4 2204.08    5133 2204.57  5270.9 2206.35
  5356.3 2213.03  5527.5 2220.06  5650.6 2230.76  5704.3 2245.98  5780.5  2247.7
#Mann= 8 ,-1 , 0
  4543.9     .16       0  4603.1     .07       0  4663.2     .16       0
  4983.8     .07       0  4995.9     .16       0    5133     .07       0
  5527.5     .16       0  5650.6     .07       0
Bank Sta=4983.8,4995.9
XS Rating Curve= 0 ,0
Exp/Cntr=0.3,0.1

Type RM Length L Ch R = 1 ,18569   ,346,346,346
BEGIN DESCRIPTION:
540
END DESCRIPTION:
XS GIS Cut Line= 3
      1509895.08      6787401.46      1509655.49       6787120.2
      1508965.97      6786672.66
#Sta/Elev= 30
  4641.8 2269.92  4708.4 2264.43  4738.1 2257.88  4743.5 2254.66  4751.2 2253.96
  4757.8 2249.29  4772.1 2246.98  4821.5 2219.27  4864.3 2208.87  4885.2 2200.13
  4921.4 2196.82  4977.4    2198  4993.3 2193.33  4993.8 2192.83  5005.4 2193.33
  5009.4 2197.34  5021.2 2198.66  5078.5 2197.39  5093.7 2202.42  5107.2 2203.91
  5171.8 2202.52  5229.5 2201.64  5338.2 2204.01    5453 2212.75  5644.1 2221.01
  5715.2 2227.68  5742.9 2231.69    5760 2236.62  5794.3    2245  5833.3 2246.35
#Mann= 7 ,-1 , 0
  4641.8     .07       0  4738.1     .16       0  4993.3     .07       0
  5005.4     .16       0  5171.8     .07       0  5644.1     .16       0
    5760     .07       0
Bank Sta=4993.3,5005.4
XS Rating Curve= 0 ,0
Exp/Cntr=0.3,0.1

Type RM Length L Ch R = 1 ,18223   ,416,416,416
BEGIN DESCRIPTION:
539
END DESCRIPTION:
XS GIS Cut Line= 3
      1510142.46      6787021.24      1509668.51      6786818.12
      1508909.08      6786597.05
#Sta/Elev= 30
  4471.2 2270.01  4488.4 2268.14  4493.9 2264.27    4541 2254.62  4593.6 2249.34
  4646.2 2248.69  4664.3 2244.84  4669.8 2239.42  4675.2 2239.96  4716.9 2223.27
  4722.4  2223.5  4740.4 2217.49  4874.4 2206.04  4950.8 2201.33  4974.4 2194.44
  4991.3 2194.11  5005.3 2190.74  5005.8 2190.24  5017.4 2190.74  5021.7 2195.96
    5069 2195.32  5183.6 2199.56  5270.2 2200.12  5328.1 2203.66  5344.6 2207.95
  5549.9 2226.72  5650.5  2239.5    5684  2246.8  5750.8 2247.35  5777.8 2252.11
#Mann= 7 ,-1 , 0
  4471.2     .07       0  4874.4     .16       0  5005.3     .07       0
  5017.4     .16       0    5069     .07       0  5270.2     .16       0
  5549.9     .07       0
Bank Sta=5005.3,5017.4
XS Rating Curve= 0 ,0
Exp/Cntr=0.3,0.1

Type RM Length L Ch R = 1 ,17807   ,184,184,184
BEGIN DESCRIPTION:
538
END DESCRIPTION:
XS GIS Cut Line= 3
      1510145.06      6786914.46      1509504.45      6786450.93
      1509033.13      6786195.74
#Sta/Elev= 30
  4207.2 2268.54  4249.1 2260.48  4291.2 2248.71  4347.7 2245.14  4362.4  2238.3
    4398 2229.11  4462.9  2221.5  4720.5 2198.92  4882.9 2197.26  4920.4 2193.49
  4948.6 2192.46  4957.2 2188.73  4963.3 2190.79  4965.8 2187.62  4966.3 2187.12
    4978 2187.62  4992.7 2192.66  5029.4  2192.5  5074.4 2192.54    5102 2208.61
    5111 2211.03  5145.7 2212.99  5183.8 2219.15  5221.8 2232.14  5227.5  2231.2
  5243.7 2236.47  5331.2 2238.62  5434.9  2251.5  5486.3  2263.5  5533.9  2280.1
#Mann= 7 ,-1 , 0
  4207.2     .16       0  4249.1     .07       0  4882.9     .16       0
  4920.4     .07       0  4965.8     .07       0    4978     .07       0
  5029.4     .16       0
Bank Sta=4965.8,4978
XS Rating Curve= 0 ,0
Exp/Cntr=0.3,0.1

Type RM Length L Ch R = 1 ,17623   ,302,302,302
BEGIN DESCRIPTION:
537
END DESCRIPTION:
XS GIS Cut Line= 3
      1510139.89      6786896.27       1509535.7      6786310.31
      1509382.05      6785784.25
#Sta/Elev= 30
  4155.5 2266.53  4178.9 2263.64  4184.8  2260.8  4214.4 2251.83  4277.9 2241.83
  4313.4 2232.45    4370 2225.58  4560.9 2207.97  4617.4 2199.79  4653.7 2197.32
  4691.7 2196.37  4751.7 2195.81  4765.9 2191.74    4780 2190.65  4842.7 2192.34
  4963.9 2191.96  4978.1  2189.3  4978.9 2187.32  4979.4 2186.82  4991.2 2187.32
  4995.2 2189.45    5001 2189.45  5030.8 2209.52  5041.2 2212.47  5114.2 2218.28
  5155.4 2226.33  5166.3  2230.3  5199.3 2235.83  5405.2 2243.06  5545.2 2257.42
#Mann= 7 ,-1 , 0
  4155.5     .16       0  4184.8     .07       0  4653.7     .16       0
  4691.7     .07       0  4842.7     .16       0  4978.9     .07       0
  4991.2     .16       0
Bank Sta=4978.9,4991.2
XS Rating Curve= 0 ,0
Exp/Cntr=0.3,0.1

Type RM Length L Ch R = 1 ,17321   ,171,171,171
BEGIN DESCRIPTION:
536
END DESCRIPTION:
XS GIS Cut Line= 3
      1510184.13      6786763.42      1509801.32      6786385.83
      1509441.94      6785755.59
#Sta/Elev= 30
  4465.9 2262.07  4469.4 2261.46  4490.4 2254.89  4497.4 2256.38  4532.8 2248.15
  4582.2 2247.36  4617.7 2234.11  4759.1 2211.71  4843.9 2200.76  4931.2 2194.55
    4957 2192.12  4986.2 2184.04  4986.7 2183.54  4998.5 2184.04  5022.4 2189.79
  5028.2 2188.03  5087.2 2192.77  5116.2 2199.67  5248.6 2205.01  5323.4 2217.83
  5372.4 2230.18  5409.9 2232.19  5415.6 2234.74  5431.5 2235.19  5447.3 2230.61
  5453.1 2233.07  5468.9 2228.47  5490.6 2234.69  5614.4 2242.77  5729.1 2257.83
#Mann= 5 ,-1 , 0
  4465.9     .16       0  4469.4     .07       0  4931.2     .16       0
  4986.2     .07       0  4998.5     .16       0
Bank Sta=4986.2,4998.5
XS Rating Curve= 0 ,0
Exp/Cntr=0.3,0.1

Type RM Length L Ch R = 1 ,17150   ,301,301,301
BEGIN DESCRIPTION:
535
END DESCRIPTION:
XS GIS Cut Line= 3
      1510285.69      6786591.55      1509939.35      6786315.51
      1509465.41      6785727.01
#Sta/Elev= 30
  4549.1 2258.24  4652.3 2247.45  4687.7 2246.76  4722.9 2243.73  4751.8 2236.41
    4787 2219.77  4793.4 2219.07  4801.4 2215.32  4886.3 2203.29  4929.5 2200.65
  4943.9 2196.38  4950.3 2192.29  4964.8  2192.7  4994.9  2182.3  4995.4  2181.8
  5007.2  2182.3  5007.5 2183.81  5021.9 2185.43  5028.3 2189.36  5085.8 2188.93
    5121 2195.53  5228.2  2199.3  5298.6  2205.7  5341.8 2212.27  5399.4  2217.3
  5533.7  2236.3  5548.1  2233.9  5655.3 2245.72  5725.7 2258.03  5747.6 2263.38
#Mann= 3 ,-1 , 0
  4549.1     .07       0  4994.9     .07       0  5007.2     .16       0
Bank Sta=4994.9,5007.2
XS Rating Curve= 0 ,0
Exp/Cntr=0.3,0.1

Type RM Length L Ch R = 1 ,16849   ,141,141,141
BEGIN DESCRIPTION:
534
END DESCRIPTION:
XS GIS Cut Line= 3
      1510499.23       6786440.5      1510007.05      6786031.66
      1509509.51      6785723.28
#Sta/Elev= 30
  4363.3 2262.09  4389.5 2260.51    4396  2257.4  4432.5 2248.29    4439 2244.23
  4488.4 2232.58  4588.7 2222.25  4638.2 2219.44  4716.3 2212.11  4850.4 2197.47
  4893.4 2194.06    4918 2188.59  4957.2 2185.81  4979.3 2185.96  5015.2 2181.55
  5015.7 2181.05  5027.5 2181.55  5029.1 2184.89  5036.8 2187.24  5042.6 2192.74
  5146.7 2198.45  5240.9 2206.39    5247 2208.14  5378.2  2224.9  5399.4 2230.62
  5420.7 2231.38  5436.1  2235.2  5551.8 2248.17  5573.1 2251.46  5588.5 2256.84
#Mann= 4 ,-1 , 0
  4363.3     .07       0    4918     .16       0  5015.2     .07       0
  5027.5     .16       0
Bank Sta=5015.2,5027.5
XS Rating Curve= 0 ,0
Exp/Cntr=0.3,0.1

Type RM Length L Ch R = 1 ,16708   ,170,170,170
BEGIN DESCRIPTION:
533
END DESCRIPTION:
XS GIS Cut Line= 3
      1510561.75      6786263.44      1510085.18      6785919.68
       1509582.6      6785643.65
#Sta/Elev= 30
    4404  2244.9    4441    2244  4455.8 2238.07  4506.1 2224.26  4541.6 2220.07
  4849.6 2200.76  4913.8 2194.15  4929.3 2192.54  4950.2 2186.61  4971.1 2185.87
  4985.8 2181.82  4994.6 2182.42  5008.5 2179.28    5009 2178.78  5020.8 2179.28
  5023.3 2184.18    5029  2184.2  5045.1 2189.82  5235.5 2198.99  5257.3 2205.98
  5300.9  2227.8    5317 2231.27  5338.8 2232.76  5354.9  2230.1  5382.4 2234.81
  5420.3 2234.02  5442.1 2236.83  5458.2 2235.39  5516.8 2243.22    5565 2250.04
#Mann= 5 ,-1 , 0
    4404     .07       0  4913.8     .16       0  5008.5     .07       0
  5020.8     .16       0  5516.8     .07       0
Bank Sta=5008.5,5020.8
XS Rating Curve= 0 ,0
Exp/Cntr=0.3,0.1

Type RM Length L Ch R = 1 ,16538   ,160,160,160
BEGIN DESCRIPTION:
532
END DESCRIPTION:
XS GIS Cut Line= 3
      1510715.42      6786185.33      1510152.89      6785768.64
      1509624.58       6785622.9
#Sta/Elev= 30
  4300.4 2252.77  4313.4 2252.33  4341.2 2246.62  4370.4 2243.15  4405.9  2242.8
  4435.2 2228.23  4462.7 2220.27  4612.5 2210.93  4691.8 2203.75  4899.7 2196.71
  4935.6 2195.24  4942.3 2191.66  4985.4  2183.9  4990.6 2178.43  4991.1 2177.93
    5003 2178.43  5008.6 2178.71  5017.7 2183.79  5070.9 2183.92  5096.8 2190.43
  5164.2 2189.55  5249.9 2194.52    5268 2201.26  5278.4 2206.52  5284.2  2211.6
  5318.6 2226.55  5340.6 2230.97  5397.7 2236.44  5486.1  2241.3  5548.5 2246.96
#Mann= 5 ,-1 , 0
  4300.4     .07       0  4899.7     .16       0  4990.6     .07       0
    5003     .16       0  5486.1     .07       0
Bank Sta=4990.6,5003
XS Rating Curve= 0 ,0
Exp/Cntr=0.3,0.1

Type RM Length L Ch R = 1 ,16378   ,304,304,304
BEGIN DESCRIPTION:
531
END DESCRIPTION:
XS GIS Cut Line= 3
       1510803.9      6786086.32       1510288.3      6785643.64
      1509619.07      6785493.19
#Sta/Elev= 30
  4234.8 2246.01  4239.5 2246.59    4275 2243.16  4311.3 2230.17    4353 2222.58
  4513.7 2206.91  4721.7 2193.38  4958.1 2189.65  4983.3  2177.3  4983.8  2176.8
  4995.7  2177.3  5006.7 2183.29  5020.3 2184.08  5061.2  2183.5  5103.5 2178.58
  5146.8 2178.15  5153.5 2182.62  5204.7 2182.33    5215 2183.86  5225.2 2188.73
    5256 2196.67  5276.5 2205.73  5281.8 2209.82  5286.9 2216.52    5297 2221.87
  5317.5 2226.17  5325.1 2229.97  5430.2 2232.74  5510.9 2240.39  5600.3 2252.57
#Mann= 7 ,-1 , 0
  4234.8     .07       0  4239.5     .16       0  4513.7     .07       0
  4958.1     .16       0  4983.3     .07       0  4995.7     .16       0
  5510.9     .07       0
#XS Ineff= 2 , 0
       0                    5020       0    2200
Permanent Ineff=
       F       F
Bank Sta=4983.3,4995.7
XS Rating Curve= 0 ,0
Exp/Cntr=0.3,0.1

Type RM Length L Ch R = 1 ,16074   ,134,134,134
BEGIN DESCRIPTION:
530
END DESCRIPTION:
XS GIS Cut Line= 3
      1510811.77      6786047.31      1510280.49      6785489.99
      1509669.29      6785253.32
#Sta/Elev= 30
  3987.6 2246.47  4027.4 2240.73  4090.9 2219.31  4213.7 2209.66  4345.7 2201.21
  4409.2 2193.21  4550.8  2189.3  4767.5 2190.62  4795.6 2188.54  4808.2 2183.96
  4832.7 2181.41  4971.7 2181.17  4982.5 2174.06    4983 2173.56  4994.9 2174.06
  5010.1 2178.01  5026.2 2175.49  5050.8 2180.97  5063.7 2185.72  5074.4 2193.43
  5080.7 2200.68    5086 2201.07  5105.3 2211.06  5110.6 2204.53  5117.3 2205.45
  5135.2  2215.5    5171 2224.38  5298.7 2241.96    5364 2254.23    5413 2254.89
#Mann= 5 ,-1 , 0
  3987.6     .16       0  4213.7     .07       0  4767.5     .16       0
  4982.5     .07       0  4994.9     .16       0
Bank Sta=4982.5,4994.9
XS Rating Curve= 0 ,0
Exp/Cntr=0.3,0.1

Type RM Length L Ch R = 1 ,15940   ,505,505,505
BEGIN DESCRIPTION:
529
END DESCRIPTION:
XS GIS Cut Line= 3
      1510986.25      6785841.57      1510129.45      6785318.12
      1509832.61       6785104.6
#Sta/Elev= 30
  3992.1 2236.64  4009.8 2236.52  4049.3  2220.9  4075.4 2214.89  4098.8 2207.75
  4134.2 2205.03  4162.7 2208.37    4184 2204.06  4391.5 2196.78    4396  2196.4
  4505.3 2190.82  4547.9    2184  4584.7 2187.94  4614.7 2183.86  4627.3 2188.92
  4694.9 2190.59  4774.3 2186.18  4788.4 2181.18  4991.1 2179.22  5000.5 2178.44
  5007.7 2172.39  5008.2 2171.89  5020.1 2172.39  5086.1 2196.36  5092.3 2203.66
  5121.7 2216.48  5210.5 2230.97    5285 2247.65  5308.3  2244.9  5361.8 2251.01
#Mann= 9 ,-1 , 0
  3992.1     .07       0  4049.3     .16       0  4075.4     .07       0
  4391.5     .16       0    4396     .07       0  4788.4     .16       0
  5007.7     .07       0  5020.1     .16       0  5210.5     .07       0
Bank Sta=5007.7,5020.1
XS Rating Curve= 0 ,0
Exp/Cntr=0.3,0.1

Type RM Length L Ch R = 1 ,15435   ,168,168,168
BEGIN DESCRIPTION:
528
END DESCRIPTION:
XS GIS Cut Line= 3
      1511056.55      6785833.76      1510556.53      6785286.87
      1509910.27       6785042.9
#Sta/Elev= 30
  4258.8 2232.76  4278.4 2231.05  4334.5 2237.97  4385.6 2229.03  4436.7 2213.08
  4476.3 2207.08  4521.7  2204.9  4653.3 2200.11  4721.2 2194.18  4793.9 2191.76
  4950.5 2185.19  4971.5 2180.99    4991 2168.39  4991.5 2167.89  5003.5 2168.39
  5014.1 2173.28  5033.5 2174.98  5140.4 2177.79  5172.5  2184.7  5247.3 2186.55
  5279.4 2194.89    5429 2209.27  5465.1 2215.22    5490 2222.91  5495.3 2220.45
  5520.1 2225.58  5525.5 2222.09    5545 2223.77  5667.1 2240.33  5690.6 2245.06
#Mann= 9 ,-1 , 0
  4258.8     .07       0  4385.6     .16       0  4436.7     .07       0
  4521.7     .16       0  4721.2     .07       0  4793.9     .16       0
    4991     .07       0  5003.5     .16       0  5667.1     .07       0
Bank Sta=4991,5003.5
XS Rating Curve= 0 ,0
Exp/Cntr=0.3,0.1

Type RM Length L Ch R = 1 ,15267   ,257,257,257
BEGIN DESCRIPTION:
527
END DESCRIPTION:
XS GIS Cut Line= 3
      1511061.72      6785266.03      1510652.89      6785156.66
      1509853.36      6785008.21
#Sta/Elev= 30
  4579.6 2231.51  4700.4 2225.73  4721.1 2219.88  4762.5 2196.06  4786.6 2189.98
    4835 2182.97  4876.4  2184.2  4917.8 2181.35  4941.6 2174.02  4969.6  2173.3
  4975.4 2166.69  4975.9 2166.19    4988 2166.69  4999.1 2173.59  5049.4 2175.01
  5112.5  2174.5  5153.2  2185.8  5366.8 2197.41  5397.3 2193.62  5404.4 2196.63
  5409.4 2194.91  5432.2 2202.78  5509.2 2210.85  5590.6 2227.64  5620.7 2229.09
  5683.7 2238.91  5712.6 2236.98  5740.7 2240.51  5789.3 2254.34    5816 2257.81
#Mann= 6 ,-1 , 0
  4579.6     .16       0  4975.4     .07       0    4988     .16       0
  5049.4     .07       0  5432.2     .16       0  5740.7     .07       0
Bank Sta=4975.4,4988
XS Rating Curve= 0 ,0
Exp/Cntr=0.3,0.1

Type RM Length L Ch R = 1 ,15010   ,300,300,300
BEGIN DESCRIPTION:
526
END DESCRIPTION:
XS GIS Cut Line= 3
      1511243.99      6785167.06      1510869.03      6784976.97
      1509838.88      6784987.38
#Sta/Elev= 30
  4516.3 2230.66  4589.8 2229.25  4706.8 2212.33    4768 2221.48  4857.1 2223.29
  4879.3 2215.61  4885.2 2209.08  4901.6 2202.48  4907.6 2195.87  4918.3 2189.05
  4923.9 2189.42  4936.1 2180.08  4960.7 2174.57  4974.4 2166.04  4974.9 2165.54
    4987 2166.04  5010.7 2172.28    5066 2172.46  5110.7 2172.05  5120.7 2175.22
  5170.7 2169.99  5200.7 2180.14  5290.7  2181.7  5550.8 2207.46  5636.9 2209.34
  5670.8 2211.63  5700.8 2223.33  5760.8 2238.02  5884.1 2242.65  5966.9 2260.66
#Mann= 6 ,-1 , 0
  4516.3     .16       0  4974.4     .07       0    4987     .16       0
    5066     .07       0  5636.9     .16       0  5884.1     .07       0
Bank Sta=4974.4,4987
XS Rating Curve= 0 ,0
Exp/Cntr=0.3,0.1

Type RM Length L Ch R = 1 ,14710   ,262,262,262
BEGIN DESCRIPTION:
525
END DESCRIPTION:
XS GIS Cut Line= 3
      1511014.87      6784927.49      1510590.39      6784794.68
      1510095.62      6784760.83
#Sta/Elev= 30
    4570 2219.01  4611.8 2216.85  4632.7 2212.19  4682.7 2207.54  4695.6 2204.25
  4737.5 2198.14  4800.4 2193.15  4810.9 2188.38  4817.8 2181.47    4823 2180.44
  4831.8 2174.87  4842.3 2172.61  4951.5 2169.86  5003.4 2163.67  5003.9 2163.17
    5016 2163.67  5020.2 2168.17  5050.2 2177.93  5090.3 2176.89  5170.5 2181.32
  5190.7 2183.85  5230.7 2192.05  5260.7 2194.96  5297.8 2202.37  5329.1 2210.79
  5334.1 2210.24    5361 2218.45  5401.1 2226.87  5421.1 2235.35  5510.7 2257.57
#Mann= 5 ,-1 , 0
    4570     .16       0  4951.5     .07       0  5003.4     .07       0
    5016     .07       0  5297.8     .16       0
Bank Sta=5003.4,5016
XS Rating Curve= 0 ,0
Exp/Cntr=0.3,0.1

Type RM Length L Ch R = 1 ,14448   ,220,220,220
BEGIN DESCRIPTION:
524
END DESCRIPTION:
XS GIS Cut Line= 3
      1511004.48        6784852.       1510660.7      6784552.49
      1510106.06      6784404.07
#Sta/Elev= 30
    4486 2204.41  4510.1 2207.42  4551.8 2199.37  4658.1 2186.75  4665.8 2188.36
  4743.6 2183.66  4800.6 2178.11  4892.7 2176.03  4921.1 2171.28  4981.4  2167.5
  5003.7 2159.43  5004.2 2158.93  5016.3 2159.43  5051.1 2168.86  5103.1 2170.45
  5131.2 2175.21  5136.4 2172.02  5154.9  2173.8  5196.3 2185.71  5206.1 2194.01
  5211.3  2191.6  5212.9 2193.55    5217 2198.56  5251.3 2202.96  5286.2 2213.45
  5361.1 2226.77  5382.6 2239.84  5446.4 2253.43  5481.3 2271.85  5516.1 2275.44
#Mann= 4 ,-1 , 0
    4486     .16       0  5003.7     .07       0  5016.3     .16       0
  5212.9     .07       0
Bank Sta=5003.7,5016.3
XS Rating Curve= 0 ,0
Exp/Cntr=0.3,0.1

Type RM Length L Ch R = 1 ,14228   ,255,255,255
BEGIN DESCRIPTION:
6
END DESCRIPTION:
XS GIS Cut Line= 3
        1511005.        6784638.      1510621.43      6784321.16
      1510505.01      6784088.01
#Sta/Elev= 30
  4502.5 2192.78  4544.8 2188.92  4608.7 2178.25  4651.7 2176.55  4686.8 2172.33
  4715.5 2171.18  4729.8 2174.44  4744.2 2173.66  4772.8 2168.81    4950 2166.24
  4964.3 2164.57  4985.1 2165.97  5006.2 2164.87  5022.2  2160.4  5022.7  2159.9
  5034.9  2160.4  5037.1  2165.6  5045.3 2168.96  5073.3 2173.44  5134.8 2187.24
  5140.4  2191.9  5148.8 2196.05  5171.2 2213.12  5179.5 2222.74  5215.9 2242.88
  5229.9 2252.17  5238.3 2260.25  5252.2 2270.51  5257.8 2274.31  5260.6 2274.31
#Mann= 3 ,-1 , 0
  4502.5     .16       0  5022.2     .07       0  5034.9     .16       0
Bank Sta=5022.2,5034.9
XS Rating Curve= 0 ,0
Exp/Cntr=0.3,0.1

Type RM Length L Ch R = 1 ,13973   ,200,200,200
BEGIN DESCRIPTION:
523
END DESCRIPTION:
XS GIS Cut Line= 3
       1511158.1      6784716.56      1510835.18      6784292.08
      1510616.44      6783906.67
#Sta/Elev= 30
  4461.6 2221.41  4520.4 2218.28  4541.2 2209.92  4594.8 2198.56  4711.8 2177.06
  4748.8 2173.75  4855.2 2171.46  4884.3 2165.85    4955 2163.35  4969.4 2158.17
  4969.9 2157.67  4982.2 2158.17  4984.1 2161.12    5027 2163.77  5080.1 2177.25
  5123.7 2181.33  5226.1 2201.42  5285.2 2225.13    5291 2230.42  5306.8 2233.68
  5312.6 2240.52  5328.5 2244.01  5334.2  2249.5    5366 2258.42  5371.7 2264.39
  5387.6 2268.03  5393.3 2274.29  5409.2  2276.6    5415 2280.55  5438.1 2282.78
#Mann= 4 ,-1 , 0
  4461.6     .07       0  4594.8     .16       0  4969.4     .07       0
  4982.2     .16       0
Bank Sta=4969.4,4982.2
XS Rating Curve= 0 ,0
Exp/Cntr=0.3,0.1

Type RM Length L Ch R = 1 ,13773   ,170,170,170
BEGIN DESCRIPTION:
522
END DESCRIPTION:
XS GIS Cut Line= 3
      1511309.11      6784583.71      1511025.28      6784266.03
      1510603.43      6783833.77
#Sta/Elev= 30
  4574.5 2213.15  4666.3 2210.93  4680.5 2207.71    4688 2204.28  4737.3 2193.13
  4779.9 2190.32  4800.9 2186.61  4883.1 2178.88  4914.5 2175.06  4957.2 2161.82
    4971 2160.96  4978.4  2156.1  4978.9  2155.6  4991.2  2156.1  4992.3 2158.67
    4997 2161.21  5041.7  2161.3  5077.1 2163.41  5105.4 2170.08  5147.9 2171.29
  5211.4 2177.67  5310.4 2191.83  5388.3 2211.91  5416.6 2221.85  5508.5 2265.88
  5515.5 2270.45  5529.6 2276.06  5543.8 2278.35  5593.3 2279.11  5604.5 2280.67
#Mann= 4 ,-1 , 0
  4574.5     .07       0  4883.1     .16       0  4978.4     .07       0
  4991.2     .16       0
Bank Sta=4978.4,4991.2
XS Rating Curve= 0 ,0
Exp/Cntr=0.3,0.1

Type RM Length L Ch R = 1 ,13603   ,141,141,141
BEGIN DESCRIPTION:
521
END DESCRIPTION:
XS GIS Cut Line= 3
      1511335.18      6784542.08       1511163.3      6784187.91
      1510655.52       6783729.6
#Sta/Elev= 30
  4596.7 2208.61  4658.4 2211.38    4698 2201.86  4743.1 2200.67  4801.3 2184.13
  4905.2 2174.14  4951.8 2160.43  4961.6 2154.39  4962.1 2153.89  4974.4 2154.39
  4987.5 2159.08    5074  2161.4  5201.8  2173.3  5392.3 2198.43  5505.9 2220.26
  5534.3 2232.62  5541.1 2232.24  5562.7 2242.52  5569.5 2242.67  5591.1 2254.44
  5597.9 2254.45  5605.3 2261.49  5612.1 2260.96  5619.5 2267.17  5626.3 2266.19
  5633.7 2271.79  5640.4 2269.79  5647.9 2274.73  5654.6 2272.61  5674.4 2275.54
#Mann= 4 ,-1 , 0
  4596.7     .07       0  4905.2     .16       0  4961.6     .07       0
  4974.4     .16       0
Bank Sta=4961.6,4974.4
XS Rating Curve= 0 ,0
Exp/Cntr=0.3,0.1

Type RM Length L Ch R = 1 ,13462   ,147,147,147
BEGIN DESCRIPTION:
519
END DESCRIPTION:
XS GIS Cut Line= 3
        1511593.      6784495.21      1511262.26      6784088.95
      1510770.11      6783539.51
#Sta/Elev= 30
  4470.6 2213.87  4488.8 2206.83  4495.2 2209.75    4567 2198.62    4623 2183.87
  4665.8 2178.01  4743.9 2174.66  4857.3 2170.64  4921.8 2167.72  4950.5 2160.09
  4985.7 2158.24  5001.2 2152.14  5001.7 2151.64    5014 2152.14  5028.6  2159.7
  5142.2 2167.75  5297.7 2190.67    5347 2192.52  5354.5 2187.31  5411.4 2192.41
  5446.5 2204.44  5453.2 2199.59  5541.8 2217.44  5630.4    2247  5637.9 2243.69
  5644.6 2246.09  5652.1 2241.12  5658.8 2245.91  5687.2 2242.11  5732.1 2253.64
#Mann= 7 ,-1 , 0
  4470.6     .07       0  4665.8     .16       0  4743.9     .07       0
  4857.3     .16       0  5001.2     .07       0    5014     .16       0
  5541.8     .07       0
Bank Sta=5001.2,5014
XS Rating Curve= 0 ,0
Exp/Cntr=0.3,0.1

Type RM Length L Ch R = 1 ,13315   ,223,223,223
BEGIN DESCRIPTION:
520
END DESCRIPTION:
XS GIS Cut Line= 3
      1511731.03      6784542.11      1511382.05      6784016.03
      1511070.12      6783342.78
#Sta/Elev= 30
  4363.6 2215.08  4500.5  2201.6  4544.4 2186.24  4565.5 2187.42  4580.5 2183.37
  4719.1 2170.81  4824.5 2163.79  4854.2  2166.6  4905.4 2159.46  4977.5 2163.02
  5004.5 2155.61  5008.3 2151.55  5008.8 2151.05  5021.2 2151.55  5027.4 2156.06
  5036.8 2157.03  5090.7 2158.28    5125 2169.12  5246.2 2187.28  5399.6 2200.06
  5479.4 2199.89    5571  2210.2  5593.9 2219.24  5599.4 2218.44  5616.8 2227.71
  5622.4 2226.03  5639.8 2235.38  5645.3 2231.18  5691.1 2240.62  5736.9 2254.66
#Mann= 4 ,-1 , 0
  4363.6     .07       0  4719.1     .16       0  5008.3     .07       0
  5021.2     .16       0
Bank Sta=5008.3,5021.2
XS Rating Curve= 0 ,0
Exp/Cntr=0.3,0.1

Type RM Length L Ch R = 1 ,13092   ,226,226,226
BEGIN DESCRIPTION:
518
END DESCRIPTION:
XS GIS Cut Line= 3
      1511749.26      6784518.69      1511574.76      6783935.31
      1511197.15      6783349.36
#Sta/Elev= 30
  4393.9 2214.11  4446.8  2206.8  4488.6 2204.86  4500.1 2202.66  4519.9  2190.6
  4540.7 2184.98  4750.9 2165.65  4775.4 2163.31  4780.8 2160.86  4808.5 2159.03
  4968.7 2155.45    4978 2148.18  4978.5 2147.68  4990.9 2148.18  5023.4 2151.17
  5029.7 2155.37  5050.8 2156.23    5072 2165.72  5081.2    2167  5087.1  2164.2
  5102.3 2169.58  5130.5 2173.69  5253.5 2183.25  5379.3  2198.1  5522.8 2209.99
  5594.4 2218.84  5637.7 2219.97  5658.8 2225.18  5679.9 2236.75  5699.9 2244.99
#Mann= 5 ,-1 , 0
  4393.9     .07       0  4750.9     .16       0    4978     .07       0
  4990.9     .16       0  5379.3     .07       0
Bank Sta=4978,4990.9
XS Rating Curve= 0 ,0
Exp/Cntr=0.3,0.1

Type RM Length L Ch R = 1 ,12866   ,155,155,155
BEGIN DESCRIPTION:
517
END DESCRIPTION:
XS GIS Cut Line= 3
      1511889.85      6784315.48       1511783.1      6783963.95
      1511270.11       6783344.2
#Sta/Elev= 30
  4629.7 2215.45  4663.6 2211.67  4696.5 2192.44  4701.7  2187.7  4736.8 2175.69
  4815.2 2166.27  4838.5 2161.96  4898.8 2160.22  4937.1 2156.96    4951 2153.25
  4975.2 2151.87  4985.9  2148.4  4986.4  2147.9  4998.8  2148.4  5020.9 2153.43
  5070.4    2157  5121.3 2163.59  5263.2 2174.15  5390.9 2187.04    5525 2195.99
  5580.5 2202.47    5667  2211.3  5703.5 2211.65  5717.8 2213.68  5724.3    2217
  5738.6 2218.33  5745.1 2221.84  5773.8 2229.55  5781.6 2230.65  5801.6 2229.46
#Mann= 4 ,-1 , 0
  4629.7     .16       0  4985.9     .07       0  4998.8     .16       0
  5580.5     .07       0
Bank Sta=4985.9,4998.8
XS Rating Curve= 0 ,0
Exp/Cntr=0.3,0.1

Type RM Length L Ch R = 1 ,12711   ,143,143,143
BEGIN DESCRIPTION:
516
END DESCRIPTION:
XS GIS Cut Line= 3
      1512163.33      6784070.74      1511889.87      6783851.97
      1511276.35      6783332.04
#Sta/Elev= 30
  4649.9 2214.62  4672.6 2215.52  4707.9  2206.9  4750.2 2184.97  4783.6 2173.48
  4992.8 2151.77  5013.6 2144.35  5014.1 2143.85  5026.6 2144.35  5027.8 2150.75
  5034.4  2151.6  5126.6 2156.41  5162.9 2163.35  5276.1 2175.98  5339.8 2178.98
  5489.2 2193.13  5538.6 2193.62  5545.2 2197.56  5552.9 2195.87  5559.5 2199.86
  5610.2 2206.74  5659.5 2207.52  5694.6 2213.65  5708.9 2212.04  5715.4 2216.43
  5723.2 2214.14  5729.7 2222.28  5737.5 2221.13  5779.9 2231.21  5804.3 2232.84
#Mann= 5 ,-1 , 0
  4649.9     .07       0  4783.6     .16       0  5013.6     .07       0
  5026.6     .16       0  5610.2     .07       0
Bank Sta=5013.6,5026.6
XS Rating Curve= 0 ,0
Exp/Cntr=0.3,0.1

Type RM Length L Ch R = 1 ,12568   ,181,181,181
BEGIN DESCRIPTION:
515
END DESCRIPTION:
XS GIS Cut Line= 3
      1512408.09      6783831.14      1511897.68      6783711.35
      1511414.24      6783342.27
#Sta/Elev= 30
  4483.2  2212.9  4578.8 2209.97  4610.6  2201.6  4647.8 2182.34    4653 2184.18
  4681.5 2177.85    4695 2179.77  4870.3 2158.65  4897.2 2151.42  4979.4 2151.31
  4989.7 2150.61    4991  2146.6  4991.5  2146.1    5004  2146.6    5040 2147.42
  5054.5 2150.57  5098.1 2149.32  5111.5 2152.61  5118.9 2158.06  5125.2  2155.9
  5133.5 2159.54  5168.8 2164.24  5268.6 2172.45  5432.8 2193.21  5476.3 2201.41
  5511.7 2215.46  5539.3 2231.62  5557.5 2235.71  5611.5  2233.5  5615.7 2235.49
#Mann= 5 ,-1 , 0
  4483.2     .07       0    4695     .16       0    4991     .07       0
    5004     .16       0  5557.5     .07       0
Bank Sta=4991,5004
XS Rating Curve= 0 ,0
Exp/Cntr=0.3,0.1

Type RM Length L Ch R = 1 ,12387   ,276,276,276
BEGIN DESCRIPTION:
514
END DESCRIPTION:
XS GIS Cut Line= 3
      1512426.36      6783807.72      1511947.16      6783547.28
      1511439.71      6783255.83
#Sta/Elev= 30
  4452.9 2212.46    4489 2213.37    4527 2209.91    4565 2197.22  4652.5 2180.58
  4821.6 2159.58    4830 2156.66  4903.3 2155.91  4919.5 2150.73    4947 2147.18
    4985  2147.9  5000.2 2143.92  5000.7 2143.42  5013.2 2143.92  5022.5 2147.78
  5044.1 2148.36  5049.9 2150.98  5242.5 2168.27  5342.5 2185.95  5402.2 2199.56
  5430.9 2210.77  5468.3 2230.67    5474 2229.52  5484.1 2233.64  5489.8 2232.16
  5505.6 2236.65  5514.5 2234.31  5548.8 2240.14  5570.4 2239.07  5583.5 2244.53
#Mann= 7 ,-1 , 0
  4452.9     .07       0  4652.5     .16       0  5000.2     .07       0
  5013.2     .16       0  5342.5     .07       0  5402.2     .16       0
  5514.5     .07       0
Bank Sta=5000.2,5013.2
XS Rating Curve= 0 ,0
Exp/Cntr=0.3,0.1

Type RM Length L Ch R = 1 ,12111   ,237,237,237
BEGIN DESCRIPTION:
513
END DESCRIPTION:
XS GIS Cut Line= 3
      1512548.67      6783448.31      1512056.53       6783307.7
      1511421.11      6783219.16
#Sta/Elev= 30
  4486.5 2208.99  4539.7 2202.23  4544.9  2204.8  4604.7 2181.43  4641.9 2173.95
  4651.5 2173.67  4667.1 2165.89  4677.5 2165.88  4685.3 2171.26  4690.5 2165.88
  4698.3 2169.85  4763.3 2164.82  4812.7 2151.36  4836.1 2148.48  4958.3 2147.23
    4990 2141.52  4990.5 2141.02    5003 2141.52  5110.9 2153.19  5171.5 2154.32
  5201.8 2164.68  5248.5 2171.59  5272.5 2178.99  5325.5 2184.33  5363.4 2186.31
  5459.5 2204.16  5524.9 2217.89    5559 2229.11  5634.7 2242.59  5639.9 2242.69
#Mann= 8 ,-1 , 0
  4486.5     .07       0  4641.9     .16       0    4990     .07       0
    5003     .16       0  5325.5     .07       0  5459.5     .16       0
    5559     .07       0  5634.7     .16       0
Bank Sta=4990,5003
XS Rating Curve= 0 ,0
Exp/Cntr=0.3,0.1
