--- Elm 01 17.prj (project) ---

Proj Title=Elm 01 17 Base Level Engineering
Current Plan=p01
Default Exp/Contr=0.3,0.1
English Units
Geom File=g01
Flow File=f01
Plan File=p01
Y Axis Title=Elevation
X Axis Title(PF)=Main Channel Distance
X Axis Title(XS)=Station
BEGIN DESCRIPTION:
Elm 01 17
END DESCRIPTION:
DSS Export Rating Curves= 0
DSS Export Rating Curve Sorted= 0
DSS Export Volume Flow Curves= 0
DXF OffsetX= 0
DXF OffsetY= 0
DXF ScaleX= 1
DXF ScaleY= 10

--- Elm 01 17.p01 (plan) ---

Plan Title=Multiple Run
Program Version=4.10
Short Identifier=Multiple
Geom File=g01
Flow File=f01
Subcritical Flow
K Sum by GR= 0
Std Step Tol= 0.01
Critical Tol= 0.01
Num of Std Step Trials= 20
Max Error Tol= 0.3
Flow Tol Ratio= 0.001
Split Flow NTrial= 30
Split Flow Tol= 0.02
Split Flow Ratio= 0.02
Log Output Level= 0
Friction Slope Method= 1
Unsteady Friction Slope Method= 2
Unsteady Bridges Friction Slope Method= 1
Parabolic Critical Depth
Global Vel Dist= 1 , 1 , 1
Global Log Level= 0
CheckData=True
Encroach Param=-1 ,0,0, 0
BEGIN DESCRIPTION:
Multiple Run
END DESCRIPTION:
Computation Interval=1HOUR
Output Interval=1HOUR
Run HTab= 0
Run UNet= 0
Run PostProcess= 0
Run WQNet= 0
UNET Theta= 1
UNET Theta Warmup= 1
UNET ZTol= 0.02
UNET ZSATol= 0.05
UNET MxIter= 20
UNET MaxInSteps= 0
UNET DtIC= 0
UNET DtMin= 0
UNET MaxCRTS= 20
UNET WFStab= 2
UNET SFStab= 1
UNET WFX= 1
UNET SFX= 1
UNET DSS MLevel= 4
UNET DZMax Abort= 100
UNET Convert EG Bridges= 0
UNET Use Existing IB Tables=-1
UNET Froude Reduction=False
UNET Froude Limit= 1
UNET Froude Power= 10
UNET Time Slicing=0,0, 5
UNET Junction Losses=0
Instantaneous Interval=1HOUR
Write IC File= 0
Write IC File at Sim End=0
Echo Input=False
Echo Parameters=False
Echo Output=False
Write Detailed= 0
WQ AD Non Conservative
WQ ULTIMATE=-1
WQ Max Comp Step=1HOUR
WQ Output Interval=15MIN
WQ Output Selected Increments= 0
WQ Output face flow=0
WQ Output face velocity=0
WQ Output face area=0
WQ Output face dispersion=0
WQ Output cell volume=0
WQ Output cell surface area=0
WQ Output cell continuity=0
WQ Output cumulative cell continuity=0
WQ Output face conc=0
WQ Output face dconc_dx=0
WQ Output face courant=0
WQ Output face peclet=0
WQ Output face adv mass=0
WQ Output face disp mass=0
WQ Output cell mass=0
WQ Output cell source sink temp=0
WQ Output cell source sink nsm=0
WQ Output MaxMinRange=-1
WQ Daily Max Min Mean=-1
WQ Daily Range=0
WQ Daily Time=0
WQ Create Restart=0
WQ Fixed Restart=0
WQ System Summary=0
WQ Use Fixed Temperature=0
Sorting and Armoring Iterations= 10
XS Update Threshold= 0.02
Hydraulics Update Threshold= 0.02
Energy Slope Method= 1
Volume Change Method= 0
XS Weighting Method= 0
Number of US Weighted Cross Sections= 1
Number of DS Weighted Cross Sections= 1
Upstream XS Weight=0.25
Main XS Weight=0.5
Downstream XS Weight=0.25
Number of DS XS's Weighted with US Boundary= 1
Upstream Boundary Weight= 1
Weight of XSs Associated with US Boundary= 0
Number of US XS's Weighted with DS Boundary= 1
Downstream Boundary Weight= 0.5
Weight of XSs Associated with DS Boundary= 0.5
Sediment Output Level= 4
Mass or Volume Output= 0
Output Increment Type= 1
Profile and TS Output Increment= 10
XS Output Flag= 0
XS Output Increment= 10
Disregard all LS=0
Disregard all Conn=0
Disregard all Breaches=0
Disregard all Pumps=0

--- Elm 01 17.f01 (steady flow) ---

Flow Title=Multiple
Number of Profiles=7
Profile Names=10-year,25-year,50-year,1pct_min,100-year,1pct_plu,500-year
River Rch & RM= Elm 01 17,Reach-1,47264
     260     368     460     287     574    1144     902
River Rch & RM= Elm 01 17,Reach-1,44043
     357     515     652     411     821    1637    1319
River Rch & RM= Elm 01 17,Reach-1,41258
     472     685     870     550    1097    2189    1768
River Rch & RM= Elm 01 17,Reach-1,32272
     510     737     931     585    1168    2330    1863
River Rch & RM= Elm 01 17,Reach-1,26072
     519     749     945     593    1184    2363    1883
River Rch & RM= Elm 01 17,Reach-1,21629
     457     644     800     493     984    1963    1510
River Rch & RM= Elm 01 17,Reach-1,15945
     519     735     916     566    1130    2254    1743
River Rch & RM= Elm 01 17,Reach-1,9052
     534     753     937     578    1153    2301    1771
River Rch & RM= Elm 01 17,Reach-1,6509
     566     801     997     616    1228    2451    1890
Boundary for River Rch & Prof#=Elm 01 17,Reach-1,1
Up Type=0
Dn Type=3
Dn Slope=0.005
Boundary for River Rch & Prof#=Elm 01 17,Reach-1,2
Up Type=0
Dn Type=3
Dn Slope=0.005
Boundary for River Rch & Prof#=Elm 01 17,Reach-1,3
Up Type=0
Dn Type=3
Dn Slope=0.005
Boundary for River Rch & Prof#=Elm 01 17,Reach-1,4
Up Type=0
Dn Type=3
Dn Slope=0.005
Boundary for River Rch & Prof#=Elm 01 17,Reach-1,5
Up Type=0
Dn Type=3
Dn Slope=0.005
Boundary for River Rch & Prof#=Elm 01 17,Reach-1,6
Up Type=0
Dn Type=3
Dn Slope=0.005
Boundary for River Rch & Prof#=Elm 01 17,Reach-1,7
Up Type=0
Dn Type=3
Dn Slope=0.005

--- Elm 01 17.g01 (geometry) ---

Geom Title=Existing Conditions

River Reach=Elm 01 17,Reach-1
Reach XY= 30
      1549639.92      6800101.92      1550505.32      6800423.28
      1551322.59      6801852.44      1551910.13      6802019.44
      1552766.79      6804748.90      1554161.21      6805395.86
      1555302.45      6806482.27      1557865.11      6807548.65
      1558465.38      6809148.22      1560227.75      6809933.65
      1560598.53      6811045.39      1560272.61      6814005.55
      1560853.11      6814443.71      1560504.89      6815108.10
      1560708.06      6816629.72      1561848.06      6817284.67
      1561462.77      6817984.59      1561962.60      6820441.33
      1562315.48      6820936.15      1562799.56      6820893.18
      1564844.24      6823228.32      1565034.34      6824368.60
      1566207.30      6824643.09      1566601.47      6824989.45
      1566560.46      6825640.45      1567341.39      6825924.75
      1568060.26      6827432.53      1568841.63      6827423.84
      1569158.53      6829486.55      1570405.00      6830988.00

Type RM Length L Ch R = 1,47264,368,368,368
BEGIN DESCRIPTION:
Elm 01 14 45.0
END DESCRIPTION:
XS GIS Cut Line= 2
      1549698.58      6800521.77      1549927.43      6800028.14
#Sta/Elev= 30
  4723.5 2000.18  4752.9 1995.45  4775.8 1993.54  4782.8 1991.89  4827.2 1987.15
  4850.1 1986.22  4918.8 1985.64  4993.1 1986.12  4998.0 1985.46  4998.3 1984.96
  5002.0 1985.46  5010.5 1986.23  5018.1 1985.71  5033.4 1986.30  5056.3 1985.46
  5061.8 1986.09  5084.7 1985.81  5102.1 1987.36  5135.8 1992.87  5158.9 1995.38
  5176.3 2000.78  5181.8 2000.73  5190.6 2004.55  5199.2 2009.41  5204.8 2007.56
  5212.6 2010.28  5222.2 2010.79  5250.6 2010.23  5256.7 2011.92  5267.6 2012.79
#Mann=5,-1,0
  4723.5    0.07       0  4998.0    0.07       0  5002.0    0.07       0
  5018.1    0.16       0  5135.8    0.07       0
Bank Sta=4998,5002
Exp/Cntr=0.3,0.1

Type RM Length L Ch R = 1,46896,355,355,355
BEGIN DESCRIPTION:
Elm 01 14 44.0
END DESCRIPTION:
XS GIS Cut Line= 3
      1549889.82      6800585.24      1550153.60      6800370.82
      1550282.27      6799925.99
#Sta/Elev= 30
  4564.1 1991.25  4572.4 1989.89  4580.4 1989.66  4622.3 1983.75  4629.9 1980.14
  4689.8 1981.17  4737.0 1983.14  4758.4 1983.30  4900.0 1983.44  4924.8 1984.52
  4930.0 1983.92  4997.2 1985.23  4998.0 1980.14  4998.3 1979.64  5002.0 1980.14
  5002.4 1984.73  5011.1 1985.68  5115.2 1989.73  5180.9 1991.36  5198.5 1992.97
  5214.5 1995.48  5219.7 1999.79  5229.7 2000.16  5240.1 1998.82  5248.1 1998.69
  5253.3 2000.64  5281.7 1998.69  5313.0 2003.47  5359.4 2005.02  5367.1 2004.41
#Mann=5,-1,0
  4564.1    0.07       0  4689.8    0.16       0  4758.4    0.07       0
  4998.0    0.07       0  5002.0    0.07       0
Bank Sta=4998,5002
Exp/Cntr=0.3,0.1

Type RM Length L Ch R = 1,46541,344,344,344
BEGIN DESCRIPTION:
Elm 01 14 43.0
END DESCRIPTION:
XS GIS Cut Line= 4
      1550137.65      6800972.50      1550255.44      6800896.12
      1550371.84      6800536.09      1550630.03      6800289.78
#Sta/Elev= 30
  4308.2 1989.31  4339.4 1989.49  4345.4 1987.06  4360.6 1989.69  4366.5 1986.95
  4375.7 1988.50  4381.7 1985.72  4396.8 1988.90  4402.8 1987.35  4412.0 1989.06
  4417.9 1986.71  4433.1 1989.66  4445.3 1986.46  4462.9 1988.53  4468.1 1986.39
  4488.7 1987.38  4500.2 1982.09  4518.9 1982.10  4526.9 1981.88  4532.2 1976.71
  4553.0 1976.70  4903.0 1977.46  4919.8 1975.07  4998.0 1974.11  4998.3 1973.61
  5002.0 1974.11  5047.2 1980.66  5068.2 1979.31  5124.8 1987.25  5183.8 1990.39
#Mann=6,-1,0
  4308.2    0.16       0  4518.9   0.033       0  4553.0    0.16       0
  4903.0    0.07       0  4998.0    0.07       0  5002.0    0.07       0
Bank Sta=4998,5002
Exp/Cntr=0.3,0.1

Type RM Length L Ch R = 1,46197,332,332,332
BEGIN DESCRIPTION:
Elm 01 14 42.0
END DESCRIPTION:
XS GIS Cut Line= 3
      1550172.67      6800962.19      1550562.90      6800814.99
      1550820.51      6800569.23
#Sta/Elev= 30
  4415.8 1989.35  4438.1 1986.26  4443.4 1990.30  4450.3 1987.10  4461.0 1984.50
  4468.3 1980.60  4473.6 1986.39  4498.5 1976.75  4503.8 1979.71  4514.5 1977.46
  4523.3 1973.86  4528.7 1976.02  4535.9 1972.34  4553.5 1971.44  4583.7 1972.25
  4803.0 1970.38  4888.9 1967.80  4922.0 1968.73  4959.7 1969.77  4998.0 1965.32
  4998.3 1964.82  5002.0 1965.32  5044.3 1967.63  5051.5 1969.13  5065.7 1968.62
  5100.9 1972.68  5108.1 1971.52  5115.0 1973.37  5122.3 1972.15  5188.9 1979.57
#Mann=4,-1,0
  4415.8    0.16       0  4922.0    0.07       0  4998.0    0.07       0
  5002.0    0.07       0
Bank Sta=4998,5002
Exp/Cntr=0.3,0.1

Type RM Length L Ch R = 1,45865,205,205,205
BEGIN DESCRIPTION:
Elm 01 14 41.0
END DESCRIPTION:
XS GIS Cut Line= 3
      1550518.73      6801066.03      1550837.25      6800997.59
      1551094.56      6800752.13
#Sta/Elev= 30
  4645.3 1964.97  4692.6 1964.07  4733.5 1964.31  4751.9 1962.53  4774.5 1962.67
  4801.3 1961.65  4876.7 1961.83  4929.3 1960.57  4976.3 1960.10  4997.4 1961.04
  4998.0 1960.10  4998.3 1959.60  5002.0 1960.10  5018.8 1961.17  5075.4 1962.11
  5096.5 1963.74  5103.7 1963.60  5132.0 1967.62  5174.5 1969.62  5181.4 1970.67
  5202.8 1971.13  5230.8 1973.34  5266.3 1973.86  5287.4 1975.22  5294.6 1974.39
  5301.5 1975.65  5308.8 1974.91  5315.7 1976.48  5322.9 1975.67  5326.7 1976.52
#Mann=4,-1,0
  4645.3    0.16       0  4929.3    0.07       0  4998.0    0.07       0
  5002.0    0.07       0
Bank Sta=4998,5002
Exp/Cntr=0.3,0.1

Type RM Length L Ch R = 1,45660,172,172,172
BEGIN DESCRIPTION:
Elm 01 14 40.0
END DESCRIPTION:
XS GIS Cut Line= 4
      1550412.70      6801396.38      1550731.23      6801327.93
      1550989.42      6801081.62      1551207.34      6800879.73
#Sta/Elev= 30
  4445.9 1969.99  4600.7 1963.19  4693.7 1961.12  4765.3 1961.36  4775.3 1960.74
  4859.1 1961.88  4873.5 1961.46  4901.5 1957.94  4943.9 1956.97  4951.2 1957.56
  4981.1 1954.73  4998.0 1954.65  4998.3 1954.15  5002.0 1954.65  5014.7 1955.39
  5028.9 1957.62  5056.5 1957.60  5149.4 1957.04  5170.4 1958.07  5177.2 1960.03
  5191.4 1961.30  5227.1 1960.84  5262.3 1961.62  5280.0 1964.77  5283.8 1965.90
  5319.0 1967.34  5326.3 1968.32  5333.2 1967.85  5396.7 1971.11  5425.6 1971.37
#Mann=7,-1,0
  4445.9    0.07       0  4859.1    0.16       0  4981.1   0.035       0
  4998.0   0.035       0  5002.0   0.035       0  5056.5    0.07       0
  5280.0   0.035       0
Bank Sta=4998,5002
Exp/Cntr=0.3,0.1

Type RM Length L Ch R = 1,45488,113,113,113
BEGIN DESCRIPTION:
Elm 01 14 39.0
END DESCRIPTION:
XS GIS Cut Line= 4
      1550499.27      6801551.09      1550817.77      6801482.65
      1551075.95      6801236.34      1551293.90      6801034.42
#Sta/Elev= 30
  4420.5 1964.64  4455.5 1963.71  4460.6 1964.20  4477.5 1962.70  4498.0 1962.63
  4509.9 1961.74  4569.6 1961.17  4598.5 1962.19  4652.9 1960.85  4682.1 1962.57
  4717.1 1959.85  4741.4 1957.93  4745.4 1958.36  4804.2 1956.69  4998.0 1949.98
  4998.3 1949.48  5002.0 1949.98  5105.6 1950.39  5179.2 1952.05  5235.9 1954.62
  5264.2 1957.20  5271.0 1959.37  5278.4 1959.56  5285.2 1961.27  5292.6 1961.17
  5299.4 1962.53  5313.5 1961.98  5320.4 1962.98  5377.1 1964.75  5400.2 1966.37
#Mann=4,-1,0
  4420.5    0.07       0  4717.1   0.035       0  4998.0   0.035       0
  5002.0   0.035       0
Bank Sta=4998,5002
Exp/Cntr=0.3,0.1

Type RM Length L Ch R = 1,45375,143,143,143
BEGIN DESCRIPTION:
Elm 01 14 38.0
END DESCRIPTION:
XS GIS Cut Line= 3
      1550707.53      6801743.22      1551190.50      6801282.48
      1551407.12      6801081.78
#Sta/Elev= 30
  4488.3 1954.59  4702.5 1956.58  4865.1 1954.80  4872.0 1953.65  4879.2 1954.69
  4886.1 1953.54  4893.4 1955.12  4900.3 1953.00  4914.5 1952.26  4921.7 1953.99
  4928.6 1951.76  4935.9 1952.51  4985.2 1949.36  4995.9 1947.22  4998.0 1946.67
  4998.3 1946.17  5002.0 1946.67  5020.8 1946.67  5041.8 1948.88  5083.1 1948.35
  5136.5 1947.82  5222.0 1950.01  5275.3 1955.94  5282.6 1958.94  5289.4 1958.26
  5296.8 1960.73  5317.8 1963.11  5362.0 1965.17  5413.8 1966.62  5451.1 1967.50
#Mann=10,-1,0
  4488.3   0.035       0  4995.9    0.07       0  4998.0    0.07       0
  5002.0    0.07       0  5083.1   0.035       0  5136.5    0.07       0
  5222.0   0.035       0  5275.3    0.07       0  5362.0   0.035       0
  5413.8    0.07       0
Bank Sta=4998,5002
Exp/Cntr=0.3,0.1

Type RM Length L Ch R = 1,45232,243,243,243
BEGIN DESCRIPTION:
Elm 01 14 37.0
END DESCRIPTION:
XS GIS Cut Line= 3
      1550797.20      6801854.60      1551280.14      6801393.87
      1551497.53      6801192.47
#Sta/Elev= 30
  4471.4 1951.56  4580.5 1952.73  4707.9 1952.01  4722.0 1952.69  4757.6 1951.72
  4764.5 1952.35  4884.6 1951.02  4920.2 1949.92  4927.1 1950.46  4976.8 1948.46
  4998.0 1944.19  4998.3 1943.69  5002.0 1944.19  5019.2 1944.40  5040.3 1946.92
  5153.6 1946.58  5174.6 1948.05  5181.9 1949.57  5188.7 1948.98  5202.9 1949.39
  5210.3 1951.32  5217.1 1951.10  5224.4 1954.25  5231.3 1951.93  5238.6 1954.60
  5245.4 1953.70  5267.0 1957.81  5287.9 1959.21  5344.6 1961.90  5435.2 1963.33
#Mann=3,-1,0
  4471.4   0.035       0  4998.0   0.035       0  5002.0   0.035       0
Bank Sta=4998,5002
Exp/Cntr=0.3,0.1

Type RM Length L Ch R = 1,44989,411,411,411
BEGIN DESCRIPTION:
Elm 01 14 36.0
END DESCRIPTION:
XS GIS Cut Line= 4
      1550901.85      6801987.42      1551205.19      6801853.67
      1551494.08      6801451.72      1551533.17      6801347.32
#Sta/Elev= 30
  4453.6 1949.89  4478.9 1950.16  4494.7 1949.49  4661.0 1946.78  4730.3 1946.90
  4736.5 1946.15  4810.5 1944.71  4816.7 1944.03  4896.5 1942.43  4911.2 1942.71
  4917.4 1941.03  4925.9 1942.72  4932.1 1942.34  4939.9 1943.29  4989.1 1943.10
  4997.1 1942.33  4998.0 1941.03  4998.3 1940.53  5001.8 1940.53  5002.0 1941.03
  5011.9 1941.21  5026.1 1942.87  5068.4 1943.32  5097.8 1945.73  5112.3 1945.74
  5118.7 1946.92  5124.8 1946.73  5161.5 1951.85  5183.7 1953.73  5391.6 1959.67
#Mann=4,-1,0
  4453.6   0.035       0  4494.7    0.07       0  4998.0    0.07       0
  5002.0    0.07       0
Bank Sta=4998,5002
Exp/Cntr=0.3,0.1

Type RM Length L Ch R = 1,44578,535,535,535
BEGIN DESCRIPTION:
Elm 01 14 35.0
END DESCRIPTION:
XS GIS Cut Line= 4
      1551029.15      6802167.59      1551367.00      6802145.93
      1551655.89      6801743.99      1551699.15      6801392.88
#Sta/Elev= 30
  4410.4 1944.74  4596.6 1941.92  4656.8 1942.09  4666.8 1941.30  4839.3 1941.60
  4981.7 1938.25  4990.3 1937.77  4996.4 1936.20  4998.0 1933.15  4998.3 1932.65
  5002.0 1933.15  5005.0 1935.05  5017.3 1933.15  5046.7 1938.24  5126.5 1938.37
  5132.7 1939.79  5147.4 1940.62  5153.6 1942.95  5162.1 1944.11  5168.3 1946.66
  5183.0 1949.51  5197.7 1950.70  5238.9 1949.42  5290.3 1949.40  5401.1 1951.06
  5471.6 1950.25  5511.9 1952.17  5519.9 1952.23  5525.0 1950.82  5597.7 1951.76
#Mann=3,-1,0
  4410.4    0.07       0  4998.0    0.07       0  5002.0    0.07       0
Bank Sta=4998,5002
Exp/Cntr=0.3,0.1

Type RM Length L Ch R = 1,44043,480,480,480
BEGIN DESCRIPTION:
Elm 01 14 34.0
END DESCRIPTION:
XS GIS Cut Line= 4
      1551380.15      6802595.93      1551787.12      6802231.44
      1552055.57      6801955.29      1552292.20      6801489.06
#Sta/Elev= 30
  4238.3 1936.68  4241.8 1936.65  4303.9 1937.18  4336.0 1935.92  4410.1 1934.61
  4487.8 1936.10  4610.4 1935.92  4641.6 1935.88  4785.9 1934.95  4842.2 1934.72
  4891.6 1930.86  4983.7 1931.68  4997.8 1931.13  4998.0 1927.40  4998.3 1926.90
  5002.0 1927.40  5004.8 1930.63  5047.2 1927.40  5061.4 1927.65  5082.5 1929.95
  5089.7 1932.41  5096.6 1931.65  5117.9 1933.49  5139.1 1931.75  5146.2 1934.42
  5169.8 1933.89  5175.9 1935.54  5234.0 1935.81  5315.1 1940.20  5692.6 1950.67
#Mann=8,-1,0
  4238.3   0.035       0  4241.8    0.07       0  4336.0   0.035       0
  4610.4    0.07       0  4641.6   0.035       0  4785.9    0.07       0
  4998.0    0.07       0  5002.0    0.07       0
Bank Sta=4998,5002
Exp/Cntr=0.3,0.1

Type RM Length L Ch R = 1,43563,400,400,400
BEGIN DESCRIPTION:
Elm 01 14 33.0
END DESCRIPTION:
XS GIS Cut Line= 4
      1551835.36      6803126.87      1552078.49      6802595.63
      1552346.94      6802319.48      1552564.81      6801537.52
#Sta/Elev= 30
  4247.9 1923.10  4330.1 1925.11  4422.2 1924.74  4433.6 1921.08  4444.6 1921.62
  4456.2 1925.01  4479.2 1923.55  4519.7 1925.30  4692.6 1926.40  4753.9 1926.26
  4812.4 1925.28  4835.0 1926.60  4877.5 1924.70  4905.8 1925.77  4969.3 1923.85
  4996.6 1924.76  4997.6 1924.86  4998.0 1921.08  4998.3 1920.58  5002.0 1921.08
  5004.8 1924.82  5033.1 1925.58  5153.2 1924.21  5467.9 1928.34  5525.9 1933.76
  5637.9 1937.02  5769.0 1938.09  5793.0 1936.73  5859.6 1940.20  6029.0 1943.80
#Mann=8,-1,0
  4247.9    0.07       0  4692.6   0.035       0  4753.9    0.07       0
  4996.6   0.035       0  4998.0   0.035       0  5002.0   0.035       0
  5637.9    0.07       0  5793.0   0.035       0
Bank Sta=4998,5002
Exp/Cntr=0.3,0.1

Type RM Length L Ch R = 1,43163,713,713,713
BEGIN DESCRIPTION:
Elm 01 14 32.0
END DESCRIPTION:
XS GIS Cut Line= 5
      1551858.34      6803195.80      1552129.14      6803105.76
      1552211.51      6802907.94      1552305.28      6802814.06
      1552653.50      6802146.69
#Sta/Elev= 30
  4440.2 1923.39  4445.5 1923.63  4450.8 1921.64  4468.3 1922.67  4499.9 1921.44
  4563.1 1921.70  4609.1 1920.87  4626.4 1919.50  4667.1 1920.50  4679.1 1920.21
  4689.6 1918.37  4698.7 1918.99  4728.2 1917.97  4752.0 1919.18  4781.3 1919.04
  4799.0 1920.44  4858.2 1919.72  4991.8 1920.64  4998.0 1917.97  4998.3 1917.47
  5002.0 1917.97  5005.9 1920.74  5106.0 1919.50  5113.2 1920.36  5226.0 1921.30
  5337.7 1924.84  5470.2 1930.99  5677.2 1935.71  5779.4 1939.80  5825.3 1939.85
#Mann=4,-1,0
  4440.2    0.07       0  4667.1   0.035       0  4998.0   0.035       0
  5002.0   0.035       0
Bank Sta=4998,5002
Exp/Cntr=0.3,0.1

Type RM Length L Ch R = 1,42450,570,570,570
BEGIN DESCRIPTION:
Elm 01 14 31.0
END DESCRIPTION:
XS GIS Cut Line= 3
      1551102.95      6803906.75      1552000.89      6803709.08
      1552809.13      6803395.72
#Sta/Elev= 30
  3677.3 1934.28  3761.3 1931.99  3913.3 1916.07  4021.4 1916.19  4065.1 1914.13
  4070.2 1916.60  4078.7 1917.21  4089.0 1914.48  4119.7 1916.36  4201.4 1913.46
  4348.0 1912.83  4391.4 1914.23  4592.5 1913.44  4794.2 1910.53  4932.0 1910.80
  4987.3 1911.86  4998.0 1909.18  4998.2 1908.68  5002.1 1909.18  5013.1 1910.22
  5040.9 1911.90  5051.2 1914.24  5056.6 1913.09  5062.3 1915.59  5067.5 1915.72
  5205.8 1923.55  5249.9 1925.41  5274.5 1929.39  5304.4 1931.77  5463.6 1937.05
#Mann=10,-1,0
  3677.3   0.035       0  3913.3    0.07       0  4391.4   0.035       0
  4592.5    0.07       0  4932.0   0.035       0  4998.0   0.035       0
  5002.1   0.035       0  5013.1    0.07       0  5067.5   0.035       0
  5205.8    0.07       0
Bank Sta=4998,5002.1
Exp/Cntr=0.3,0.1

Type RM Length L Ch R = 1,41880,622,622,622
BEGIN DESCRIPTION:
Elm 01 14 30.0
END DESCRIPTION:
XS GIS Cut Line= 3
      1551153.43      6804399.57      1552176.20      6804481.66
      1552826.79      6803682.05
#Sta/Elev= 30
  3512.3 1922.89  3704.5 1917.39  3774.7 1918.82  3838.3 1917.31  3905.1 1914.66
  3925.2 1915.69  4125.8 1911.56  4308.3 1903.51  4416.8 1900.70  4426.0 1902.87
  4477.0 1901.06  4554.9 1903.32  4768.6 1904.81  4890.9 1906.13  4977.2 1904.85
  4994.4 1904.81  4998.0 1900.70  4998.2 1900.20  5002.1 1900.70  5002.3 1904.65
  5123.2 1903.71  5151.0 1905.41  5158.9 1908.35  5187.6 1907.00  5214.9 1910.14
  5237.2 1908.69  5272.3 1912.63  5329.5 1915.36  5528.0 1921.06  5569.2 1923.79
#Mann=7,-1,0
  3512.3    0.07       0  3838.3   0.035       0  4768.6    0.07       0
  4890.9   0.035       0  4977.2    0.07       0  4998.0    0.07       0
  5002.1    0.07       0
Bank Sta=4998,5002.1
Exp/Cntr=0.3,0.1

Type RM Length L Ch R = 1,41258,608,608,608
BEGIN DESCRIPTION:
Elm 01 14 29.0
END DESCRIPTION:
XS GIS Cut Line= 3
      1551989.79      6805709.08      1552651.16      6804735.61
      1553333.50      6803873.82
#Sta/Elev= 30
  3722.3 1949.42  3741.1 1948.98  3756.0 1943.67  3827.9 1933.28  4001.5 1932.25
  4100.4 1915.89  4259.1 1896.83  4504.5 1896.95  4519.5 1894.55  4533.6 1897.22
  4735.0 1896.00  4851.0 1898.85  4938.1 1898.98  4992.9 1898.81  4997.9 1894.55
  4998.2 1894.05  5002.2 1894.55  5007.3 1898.47  5021.8 1899.66  5190.8 1899.97
  5359.6 1900.19  5392.0 1900.19  5433.6 1910.29  5491.3 1907.60  5497.7 1909.76
  5541.0 1904.40  5648.4 1906.85  5912.8 1924.75  5915.8 1925.24  5998.4 1930.91
#Mann=9,-1,0
  3722.3    0.07       0  4851.0   0.035       0  4938.1    0.07       0
  4997.9    0.07       0  5002.2    0.07       0  5190.8   0.035       0
  5359.6    0.07       0  5912.8   0.035       0  5915.8    0.07       0
Bank Sta=4997.9,5002.2
Exp/Cntr=0.3,0.1

Type RM Length L Ch R = 1,40650,483,483,483
BEGIN DESCRIPTION:
Elm 01 14 28.0
END DESCRIPTION:
XS GIS Cut Line= 3
      1552654.98      6805788.04      1553201.97      6804983.95
      1553669.81      6804422.79
#Sta/Elev= 30
  4027.5 1929.03  4154.9 1919.93  4165.9 1919.15  4322.6 1909.71  4445.1 1903.53
  4451.1 1899.92  4466.1 1897.51  4495.9 1895.37  4552.8 1898.29  4582.7 1895.30
  4732.4 1892.68  4834.2 1895.15  4849.6 1892.08  4941.9 1892.86  4996.8 1889.66
  4997.3 1889.16  5003.2 1889.66  5027.7 1893.34  5078.3 1892.31  5212.8 1893.67
  5263.8 1894.47  5336.4 1895.14  5475.5 1895.60  5553.6 1906.08  5584.0 1914.00
  5623.9 1923.39  5652.5 1934.41  5681.1 1941.18  5709.8 1943.78  5730.6 1940.93
#Mann=12,-1,0
  4027.5   0.035       0  4154.9    0.07       0  4165.9   0.035       0
  4322.6    0.07       0  4849.6    0.16       0  4996.8    0.07       0
  5003.2    0.16       0  5078.3   0.035       0  5212.8    0.07       0
  5263.8   0.035       0  5336.4    0.07       0  5584.0    0.16       0
Bank Sta=4996.8,5003.2
Exp/Cntr=0.3,0.1

Type RM Length L Ch R = 1,40167,472,472,472
BEGIN DESCRIPTION:
Elm 01 14 27.0
END DESCRIPTION:
XS GIS Cut Line= 3
      1553004.99      6805988.01      1553575.16      6805187.76
      1554257.03      6804057.51
#Sta/Elev= 30
  4017.4 1922.88  4156.1 1916.27  4263.9 1912.21  4378.0 1908.53  4407.1 1906.96
  4591.9 1900.75  4605.1 1900.06  4844.8 1892.50  4900.1 1890.71  4921.0 1887.14
  4956.7 1890.22  4992.3 1889.60  4996.8 1887.12  4997.3 1886.62  5003.3 1887.12
  5028.8 1890.01  5145.3 1890.72  5160.8 1887.57  5188.0 1891.07  5258.1 1890.79
  5494.7 1891.42  5626.7 1905.27  5662.9 1906.52  5669.4 1904.23  5793.9 1901.79
  5875.2 1910.55  5982.9 1905.54  6120.9 1906.04  6214.9 1912.31  6320.0 1932.47
#Mann=13,-1,0
  4017.4    0.07       0  4156.1   0.035       0  4263.9    0.07       0
  4378.0   0.035       0  4407.1    0.07       0  4591.9   0.035       0
  4605.1    0.07       0  4844.8    0.16       0  4996.8    0.07       0
  5003.3    0.16       0  5258.1    0.07       0  5662.9   0.035       0
  5982.9    0.07       0
Bank Sta=4996.8,5003.3
Exp/Cntr=0.3,0.1

Type RM Length L Ch R = 1,39695,116,116,116
BEGIN DESCRIPTION:
Elm 01 14 26.0
END DESCRIPTION:
XS GIS Cut Line= 5
      1553636.81      6806242.44      1554009.16      6805602.52
      1553993.56      6805328.32      1553988.03      6805132.40
      1554406.17      6804457.08
#Sta/Elev= 30
  3997.9 1918.98  4028.0 1914.57  4037.7 1912.18  4043.8 1908.24  4049.6 1909.74
  4059.5 1906.74  4072.5 1908.09  4102.5 1904.18  4167.1 1899.33  4225.8 1900.73
  4305.4 1899.00  4339.4 1897.85  4546.9 1890.97  4717.3 1887.51  4738.0 1883.65
  4997.3 1883.00  5033.2 1884.26  5053.2 1888.98  5083.3 1891.09  5123.3 1887.62
  5209.4 1889.22  5247.1 1887.29  5322.7 1888.77  5508.2 1890.34  5544.9 1890.77
  5943.3 1899.47  5972.6 1902.47  5978.6 1905.29  5988.0 1906.60  6003.2 1906.19
#Mann=9,-1,0
  3997.9    0.07       0  4305.4   0.035       0  4339.4    0.07       0
  4738.0    0.04       0  5033.2    0.07       0  5209.4    0.16       0
  5322.7    0.07       0  5508.2   0.035       0  5544.9    0.07       0
Bank Sta=4738,5033.2
Exp/Cntr=0.3,0.1

Type RM Length L Ch R = 1,39579,404,404,404
BEGIN DESCRIPTION:
Elm 01 14 25.4
END DESCRIPTION:
XS GIS Cut Line= 5
      1553885.79      6806366.71      1554147.48      6805771.80
      1554122.02      6805437.15      1554029.04      6805263.73
      1554532.35      6804442.15
#Sta/Elev= 30
  3958.7 1918.29  3989.3 1914.88  4001.0 1910.21  4018.1 1910.41  4077.5 1903.66
  4228.8 1898.17  4296.7 1896.78  4314.6 1898.21  4320.1 1896.68  4361.3 1899.92
  4395.5 1895.41  4435.5 1893.08  4569.9 1887.21  4608.0 1890.25  4789.3 1891.78
  4812.8 1891.72  4903.3 1892.94  4953.1 1889.64  4996.7 1887.14  4997.2 1886.64
  5003.3 1887.14  5052.7 1891.07  5130.2 1891.87  5151.8 1891.52  5215.8 1887.25
  5404.7 1888.53  5732.3 1892.61  5979.8 1902.14  6095.9 1908.83  6104.5 1910.93
#Mann=11,-1,0
  3958.7    0.07       0  4228.8   0.035       0  4435.5    0.07       0
  4789.3    0.16       0  4812.8    0.07       0  4953.1    0.16       0
  4996.7    0.07       0  5003.3    0.16       0  5130.2    0.07       0
  5151.8    0.16       0  5404.7    0.07       0
Bank Sta=4996.7,5003.3
Exp/Cntr=0.3,0.1

Type RM Length L Ch R = 1,39175,456,456,456
BEGIN DESCRIPTION:
Elm 01 14 25.0
END DESCRIPTION:
XS GIS Cut Line= 3
      1554095.46      6806200.11      1554195.51      6805742.68
      1554754.98      6804838.04
#Sta/Elev= 30
  4448.1 1901.13  4501.4 1903.22  4560.3 1900.25  4593.7 1900.89  4634.5 1895.52
  4653.2 1890.85  4729.4 1889.24  4808.5 1888.10  4838.9 1890.04  4844.0 1887.40
  4859.7 1885.42  4941.7 1886.14  4996.7 1879.68  4997.2 1879.18  5003.3 1879.68
  5005.5 1880.94  5020.9 1879.68  5042.1 1883.56  5060.2 1884.54  5276.2 1885.28
  5357.2 1885.27  5414.5 1883.24  5502.7 1883.83  5560.3 1884.83  5667.4 1885.33
  5719.4 1888.69  5757.1 1888.11  5862.5 1889.57  5958.6 1894.42  5980.0 1896.36
#Mann=12,-1,0
  4448.1    0.07       0  4593.7   0.035       0  4729.4    0.07       0
  4996.7    0.07       0  5003.3    0.07       0  5060.2    0.16       0
  5276.2    0.07       0  5357.2    0.16       0  5502.7    0.07       0
  5560.3    0.16       0  5757.1    0.07       0  5958.6    0.16       0
Bank Sta=4996.7,5003.3
Exp/Cntr=0.3,0.1

Type RM Length L Ch R = 1,38719,386,386,386
BEGIN DESCRIPTION:
Elm 01 14 24.0
END DESCRIPTION:
XS GIS Cut Line= 3
      1554305.03      6806137.98      1554639.96      6805838.35
      1554955.00      6804638.00
#Sta/Elev= 30
  4550.6 1894.74  4628.7 1889.15  4876.9 1884.08  4975.6 1882.10  4996.7 1877.68
  4997.2 1877.18  5003.3 1877.68  5010.7 1879.79  5038.0 1882.74  5124.4 1884.46
  5134.8 1882.73  5154.0 1883.89  5391.1 1882.95  5436.6 1881.64  5708.9 1886.42
  5734.4 1888.42  5750.6 1887.30  5765.4 1888.53  5854.9 1889.98  5981.2 1892.96
  6013.5 1892.56  6096.3 1896.31  6102.3 1895.55  6107.4 1897.51  6137.5 1898.47
  6142.7 1900.43  6183.0 1905.15  6218.2 1905.38  6223.4 1907.42  6241.0 1907.11
#Mann=6,-1,0
  4550.6    0.07       0  4876.9    0.16       0  4996.7    0.07       0
  5003.3    0.16       0  5750.6   0.035       0  5854.9    0.07       0
Bank Sta=4996.7,5003.3
Exp/Cntr=0.3,0.1

Type RM Length L Ch R = 1,38333,420,420,420
BEGIN DESCRIPTION:
Elm 01 14 23.0
END DESCRIPTION:
XS GIS Cut Line= 3
      1554234.63      6806877.11      1554851.27      6806265.09
      1555254.99      6804938.04
#Sta/Elev= 30
  3946.7 1892.74  4032.6 1890.57  4203.0 1882.70  4307.0 1880.21  4391.8 1883.12
  4451.6 1881.48  4589.5 1881.97  4595.0 1881.96  4738.3 1884.47  4801.9 1891.99
  4854.3 1883.63  4950.5 1878.97  4969.2 1878.45  4983.9 1874.60  4989.0 1876.58
  4996.7 1874.60  4997.2 1874.10  5003.3 1874.60  5022.0 1880.21  5052.0 1877.43
  5153.5 1880.80  5408.3 1882.91  5559.7 1881.06  5622.7 1881.42  5965.8 1884.44
  6094.4 1886.32  6121.9 1886.93  6153.4 1889.35  6171.3 1894.38  6202.6 1895.35
#Mann=17,-1,0
  3946.7    0.07       0  4032.6   0.035       0  4203.0    0.07       0
  4451.6   0.035       0  4589.5    0.07       0  4595.0   0.035       0
  4950.5    0.07       0  4989.0    0.16       0  4996.7    0.07       0
  5003.3    0.16       0  5052.0    0.07       0  5153.5    0.16       0
  5559.7    0.07       0  5622.7    0.16       0  5965.8    0.07       0
  6094.4   0.035       0  6121.9    0.07       0
Bank Sta=4996.7,5003.3
Exp/Cntr=0.3,0.1

Type RM Length L Ch R = 1,37913,571,571,571
BEGIN DESCRIPTION:
Elm 01 14 22.0
END DESCRIPTION:
XS GIS Cut Line= 3
      1555287.16      6807218.32      1555123.71      6806642.51
      1555672.84      6804665.41
#Sta/Elev= 30
  4087.8 1912.90  4108.9 1914.31  4114.1 1911.88  4148.0 1911.15  4153.2 1908.22
  4192.3 1901.93  4266.3 1893.92  4338.3 1886.48  4464.1 1881.04  4492.2 1879.95
  4594.8 1877.28  4812.9 1873.89  4934.7 1876.50  4973.9 1877.29  4996.7 1872.46
  4997.2 1871.96  5003.4 1872.46  5013.4 1875.63  5210.0 1877.43  5251.5 1880.08
  5504.3 1879.92  5605.1 1879.60  5676.6 1877.50  5697.8 1880.16  5757.7 1879.46
  5806.9 1879.53  6210.4 1883.64  6528.0 1888.58  6576.5 1892.23  6738.3 1893.00
#Mann=15,-1,0
  4087.8   0.035       0  4114.1    0.07       0  4266.3   0.035       0
  4464.1    0.07       0  4492.2   0.035       0  4594.8    0.16       0
  4812.9    0.07       0  4934.7    0.16       0  4996.7    0.07       0
  5003.4    0.16       0  5504.3    0.07       0  5605.1    0.16       0
  5757.7    0.07       0  5806.9    0.16       0  6210.4    0.07       0
Bank Sta=4996.7,5003.4
Exp/Cntr=0.3,0.1

Type RM Length L Ch R = 1,37342,489,489,489
BEGIN DESCRIPTION:
Elm 01 14 21.0
END DESCRIPTION:
XS GIS Cut Line= 3
      1555455.02      6806937.96      1555653.35      6806542.39
      1556330.21      6804638.00
#Sta/Elev= 30
  4557.5 1886.96  4622.6 1880.27  4669.1 1877.01  4736.4 1872.55  4758.8 1873.55
  4781.2 1877.77  4839.5 1875.59  4878.6 1878.38  4945.6 1871.93  4993.3 1871.76
  4996.5 1871.76  4997.0 1871.26  5003.6 1871.76  5031.1 1871.91  5068.3 1872.53
  5076.6 1875.34  5089.6 1876.32  5229.0 1876.17  5348.9 1876.12  5386.7 1880.12
  5397.3 1877.87  5429.2 1876.81  5441.5 1879.33  5503.5 1876.17  5567.1 1878.02
  5692.1 1875.88  5817.2 1877.24  6348.6 1881.36  6751.1 1887.17  7021.1 1894.77
#Mann=11,-1,0
  4557.5   0.035       0  4622.6    0.07       0  4669.1   0.035       0
  4993.3    0.16       0  4996.5    0.07       0  5003.6    0.16       0
  5031.1    0.07       0  5229.0    0.16       0  5692.1    0.07       0
  5817.2    0.16       0  6348.6    0.07       0
Bank Sta=4996.5,5003.6
Exp/Cntr=0.3,0.1

Type RM Length L Ch R = 1,36853,478,478,478
BEGIN DESCRIPTION:
Elm 01 14 20.0
END DESCRIPTION:
XS GIS Cut Line= 3
      1555655.03      6807037.97      1556052.81      6806631.82
      1556655.00      6805438.00
#Sta/Elev= 30
  4431.5 1890.70  4466.8 1884.42  4543.5 1876.84  4608.3 1873.54  4735.6 1873.12
  4742.6 1868.56  4763.9 1867.58  4770.9 1871.00  4778.0 1868.05  4785.0 1871.15
  4792.1 1869.09  4799.1 1873.38  4820.4 1873.69  4990.2 1872.18  4996.5 1867.58
  4997.0 1867.08  5003.6 1867.58  5004.9 1872.20  5080.1 1872.43  5188.3 1872.68
  5283.9 1872.99  5299.3 1872.94  5386.1 1873.31  5528.8 1875.04  5698.7 1874.06
  5817.9 1875.43  5933.9 1878.92  6061.1 1887.19  6306.0 1895.38  6337.1 1896.28
#Mann=12,-1,0
  4431.5    0.07       0  4543.5    0.16       0  4996.5    0.07       0
  5003.6    0.16       0  5080.1    0.07       0  5188.3   0.035       0
  5283.9    0.07       0  5299.3   0.035       0  5386.1    0.07       0
  5528.8    0.16       0  5817.9    0.07       0  6306.0   0.035       0
Bank Sta=4996.5,5003.6
Exp/Cntr=0.3,0.1

Type RM Length L Ch R = 1,36375,435,435,435
BEGIN DESCRIPTION:
Elm 01 14 19.0
END DESCRIPTION:
XS GIS Cut Line= 3
      1555999.66      6807563.85      1556430.90      6806815.04
      1556796.01      6805761.94
#Sta/Elev= 30
  4135.9 1906.62  4254.5 1901.02  4276.1 1895.56  4281.9 1892.44  4362.3 1883.89
  4533.3 1877.59  4554.8 1874.22  4560.6 1875.35  4576.4 1871.56  4594.7 1870.61
  4650.4 1866.70  4715.8 1869.15  4780.4 1866.76  4839.3 1873.24  4855.1 1869.95
  4860.9 1871.54  4869.6 1869.29  4898.1 1869.79  4994.5 1870.41  4996.1 1866.70
  4996.6 1866.20  5004.0 1866.70  5007.5 1870.24  5051.9 1870.68  5326.5 1871.42
  5606.6 1873.95  5833.0 1873.44  5949.4 1877.19  6063.1 1884.94  6114.6 1886.47
#Mann=7,-1,0
  4135.9   0.035       0  4594.7    0.07       0  4898.1    0.16       0
  4996.1    0.07       0  5004.0    0.16       0  5051.9   0.035       0
  5326.5    0.07       0
Bank Sta=4996.1,5004
Exp/Cntr=0.3,0.1

Type RM Length L Ch R = 1,35940,480,480,480
BEGIN DESCRIPTION:
Elm 01 14 18.0
END DESCRIPTION:
XS GIS Cut Line= 3
      1556505.00      6807488.00      1556710.86      6807085.93
      1557805.00      6805888.00
#Sta/Elev= 30
  4548.3 1878.57  4568.1 1878.84  4702.5 1873.54  4785.1 1870.82  4972.9 1865.89
  4996.0 1861.40  4996.5 1860.90  5004.0 1861.40  5025.1 1862.47  5037.1 1862.78
  5043.9 1866.05  5067.1 1865.43  5086.5 1864.74  5100.7 1861.73  5121.6 1864.94
  5383.7 1868.11  5971.5 1868.91  6008.6 1867.16  6041.8 1869.09  6112.7 1866.53
  6190.4 1875.10  6260.9 1875.37  6307.1 1877.11  6367.4 1881.31  6389.0 1880.45
  6423.7 1884.74  6480.9 1888.16  6558.6 1898.66  6586.9 1897.70  6622.4 1891.69
#Mann=12,-1,0
  4548.3   0.035       0  4568.1    0.07       0  4702.5   0.035       0
  4785.1    0.07       0  4996.0    0.07       0  5004.0    0.07       0
  5025.1    0.16       0  5067.1    0.07       0  6008.6    0.16       0
  6260.9    0.07       0  6307.1   0.035       0  6423.7    0.07       0
Bank Sta=4996,5004
Exp/Cntr=0.3,0.1

Type RM Length L Ch R = 1,35460,437,437,437
BEGIN DESCRIPTION:
Elm 01 14 17.0
END DESCRIPTION:
XS GIS Cut Line= 3
      1556804.98      6807588.02      1557077.24      6807310.59
      1557755.01      6806087.99
#Sta/Elev= 30
  4611.3 1884.36  4618.4 1883.37  4632.5 1876.01  4646.7 1872.94  4858.8 1865.18
  4964.9 1863.78  4986.1 1860.20  4993.1 1862.46  4996.0 1860.20  4996.5 1859.70
  5004.1 1860.20  5007.2 1863.72  5014.4 1863.80  5050.7 1861.98  5278.5 1865.53
  5940.5 1868.38  6015.6 1866.92  6134.6 1873.01  6156.4 1875.18  6162.1 1878.17
  6169.2 1875.43  6192.1 1880.30  6199.9 1879.57  6205.6 1882.68  6221.6 1881.71
  6243.4 1886.51  6259.4 1885.13  6293.1 1886.17  6346.4 1891.55  6397.9 1893.04
#Mann=4,-1,0
  4611.3    0.07       0  4996.0    0.07       0  5004.1    0.07       0
  6293.1   0.035       0
Bank Sta=4996,5004.1
Exp/Cntr=0.3,0.1

Type RM Length L Ch R = 1,35023,446,446,446
BEGIN DESCRIPTION:
Elm 01 14 16.0
END DESCRIPTION:
XS GIS Cut Line= 3
      1556905.01      6807937.99      1557456.88      6807387.48
      1557755.01      6806187.97
#Sta/Elev= 30
  4220.5 1892.50  4319.5 1884.68  4425.5 1872.63  4489.2 1869.25  4637.7 1863.36
  4658.9 1865.31  4786.2 1861.21  4807.4 1862.68  4828.6 1858.94  4849.8 1863.06
  4906.4 1860.60  4991.2 1861.74  4995.9 1858.94  4996.4 1858.44  5004.1 1858.94
  5008.8 1861.51  5020.1 1861.85  5386.0 1864.95  5566.2 1863.96  5895.9 1867.78
  5957.8 1866.17  5999.0 1868.80  6047.4 1875.58  6102.0 1875.47  6130.0 1879.56
  6135.2 1877.40  6171.4 1886.50  6176.5 1884.79  6232.8 1891.35  6236.0 1891.37
#Mann=4,-1,0
  4220.5    0.07       0  4995.9    0.07       0  5004.1    0.07       0
  6232.8   0.035       0
Bank Sta=4995.9,5004.1
Exp/Cntr=0.3,0.1

Type RM Length L Ch R = 1,34577,467,467,467
BEGIN DESCRIPTION:
Elm 01 14 15.0
END DESCRIPTION:
XS GIS Cut Line= 3
      1557455.02      6808137.97      1557798.97      6807529.80
      1558405.00      6806738.00
#Sta/Elev= 30
  4301.3 1889.56  4305.0 1889.51  4352.0 1887.36  4462.1 1871.25  4498.3 1867.95
  4638.3 1863.08  4749.3 1861.14  4772.3 1857.46  4778.3 1858.67  4784.1 1862.27
  4794.2 1863.31  4829.7 1858.47  4837.5 1860.84  4888.4 1860.50  4990.6 1860.53
  4995.9 1857.46  4996.4 1856.96  5004.1 1857.46  5005.1 1859.65  5073.3 1859.37
  5119.4 1858.78  5148.4 1860.53  5169.2 1858.33  5228.9 1860.06  5462.1 1862.55
  5555.6 1861.63  5796.7 1863.10  5940.0 1872.06  5989.8 1877.15  5997.1 1879.53
#Mann=7,-1,0
  4301.3    0.07       0  4305.0   0.035       0  4888.4    0.07       0
  4995.9    0.07       0  5004.1    0.07       0  5073.3    0.16       0
  5228.9    0.07       0
Bank Sta=4995.9,5004.1
Exp/Cntr=0.3,0.1

Type RM Length L Ch R = 1,34110,446,446,446
BEGIN DESCRIPTION:
Elm 01 14 14.0
END DESCRIPTION:
XS GIS Cut Line= 3
      1557504.99      6808138.01      1557848.82      6807885.81
      1558890.52      6806949.88
#Sta/Elev= 30
  4573.6 1887.85  4580.9 1888.19  4637.3 1878.00  4645.8 1875.00  4681.3 1870.17
  4839.5 1863.22  4967.2 1859.06  4995.7 1856.46  4996.2 1855.96  5004.4 1856.46
  5038.0 1859.65  5286.2 1857.48  5371.3 1860.09  5438.1 1859.48  5547.8 1859.80
  5576.2 1857.99  5590.4 1859.37  5618.8 1858.31  5816.9 1861.00  5873.7 1860.64
  5887.9 1858.88  5909.0 1861.08  5951.5 1860.43  6043.5 1863.15  6108.5 1866.97
  6157.0 1872.84  6185.4 1879.08  6199.6 1879.91  6348.6 1878.37  6400.4 1876.90
#Mann=8,-1,0
  4573.6   0.035       0  4839.5    0.07       0  4967.2   0.035       0
  4995.7   0.035       0  5004.4   0.035       0  5438.1    0.07       0
  6108.5   0.035       0  6348.6    0.07       0
Bank Sta=4995.7,5004.4
Exp/Cntr=0.3,0.1

Type RM Length L Ch R = 1,33664,480,480,480
BEGIN DESCRIPTION:
Elm 01 14 13.0
END DESCRIPTION:
XS GIS Cut Line= 3
      1557755.04      6808487.97      1558031.05      6808265.19
      1558855.03      6807537.97
#Sta/Elev= 30
  4645.3 1886.31  4673.3 1884.45  4702.0 1878.65  4716.4 1873.69  4730.8 1870.67
  4745.2 1868.22  4758.8 1867.31  4865.2 1860.95  4951.5 1858.08  4986.7 1853.92
  4993.1 1855.48  4995.6 1853.92  4996.1 1853.42  5004.4 1853.92  5007.6 1856.20
  5015.2 1857.34  5036.1 1857.04  5043.6 1858.18  5631.8 1857.29  5783.5 1858.31
  5858.5 1858.26  5893.6 1859.38  6012.5 1858.24  6042.5 1858.79  6056.7 1861.25
  6063.4 1863.55  6070.9 1864.59  6091.8 1874.11  6095.6 1876.72  6099.0 1876.72
#Mann=6,-1,0
  4645.3   0.035       0  4758.8    0.07       0  4995.6    0.07       0
  5004.4    0.07       0  5783.5   0.035       0  6012.5    0.07       0
Bank Sta=4995.6,5004.4
Exp/Cntr=0.3,0.1

Type RM Length L Ch R = 1,33184,912,912,912
BEGIN DESCRIPTION:
Elm 01 14 12.0
END DESCRIPTION:
XS GIS Cut Line= 3
      1557904.97      6808838.02      1558282.14      6808564.16
      1559105.03      6807837.97
#Sta/Elev= 30
  4533.9 1882.16  4562.1 1880.42  4602.7 1873.02  4723.2 1864.20  4855.2 1857.47
  4985.0 1856.39  4991.2 1856.06  4995.6 1851.68  4996.1 1851.18  5004.4 1851.68
  5006.1 1855.34  5027.9 1851.68  5034.6 1855.81  5042.1 1856.47  5148.4 1855.71
  5169.3 1853.27  5190.5 1856.31  5271.5 1856.20  5285.6 1856.04  5537.3 1855.36
  5679.6 1856.22  5906.3 1854.84  5941.4 1855.69  6026.8 1861.93  6055.2 1866.05
  6076.1 1867.29  6083.7 1870.15  6090.3 1870.00  6094.1 1873.10  6097.5 1873.10
#Mann=7,-1,0
  4533.9    0.07       0  4602.7   0.035       0  4723.2    0.07       0
  4995.6    0.07       0  5004.4    0.07       0  5271.5   0.035       0
  5285.6    0.07       0
Bank Sta=4995.6,5004.4
Exp/Cntr=0.3,0.1

Type RM Length L Ch R = 1,32272,479,479,479
BEGIN DESCRIPTION:
Elm 01 14 11.0
END DESCRIPTION:
XS GIS Cut Line= 3
      1558084.39      6809290.86      1558564.19      6809317.63
      1559307.67      6808172.58
#Sta/Elev= 30
  4325.8 1872.87  4362.9 1875.65  4456.6 1876.73  4506.7 1870.38  4526.7 1865.55
  4536.7 1867.27  4606.9 1868.42  4646.9 1865.35  4677.0 1857.56  4715.8 1856.36
  4799.9 1855.70  4944.3 1855.23  4972.8 1853.28  4980.5 1850.80  4986.5 1851.17
  4995.5 1847.65  4996.0 1847.15  5004.5 1847.65  5053.0 1854.39  5515.1 1850.70
  5580.9 1852.76  5883.5 1852.42  6013.4 1854.05  6057.8 1856.28  6085.8 1860.10
  6101.0 1864.89  6122.1 1866.71  6137.2 1871.25  6158.3 1870.73  6171.6 1873.77
#Mann=5,-1,0
  4325.8    0.07       0  4715.8   0.035       0  4799.9    0.07       0
  4995.5    0.07       0  5004.5    0.07       0
Bank Sta=4995.5,5004.5
Exp/Cntr=0.3,0.1

Type RM Length L Ch R = 1,31793,485,485,485
BEGIN DESCRIPTION:
Elm 01 14 10.0
END DESCRIPTION:
XS GIS Cut Line= 3
      1558418.57      6810146.91      1559437.96      6808754.96
      1559426.10      6808256.01
#Sta/Elev= 30
  4073.1 1874.61  4308.0 1868.57  4427.1 1864.18  4448.8 1864.94  4463.5 1864.27
  4469.7 1861.91  4605.6 1857.60  4670.4 1853.59  4784.1 1851.19  4826.0 1851.47
  4903.1 1851.93  4977.7 1850.49  4992.3 1849.00  4995.5 1846.03  4996.0 1845.53
  5004.5 1846.03  5027.4 1849.52  5057.2 1852.32  5123.6 1851.72  5379.2 1850.68
  5429.3 1848.57  5450.1 1851.16  5498.2 1850.33  5555.5 1850.67  5624.7 1850.45
  5736.5 1849.23  6068.7 1851.91  6164.2 1857.55  6245.5 1862.59  6297.5 1861.99
#Mann=16,-1,0
  4073.1    0.07       0  4308.0   0.035       0  4427.1    0.07       0
  4784.1   0.035       0  4826.0    0.07       0  4903.1   0.035       0
  4995.5   0.035       0  5004.5   0.035       0  5027.4   0.035       0
  5123.6    0.07       0  5379.2   0.035       0  5498.2    0.07       0
  5555.5   0.035       0  5624.7    0.07       0  6068.7   0.035       0
  6164.2    0.07       0
Bank Sta=4995.5,5004.5
Exp/Cntr=0.3,0.1

Type RM Length L Ch R = 1,31308,553,553,553
BEGIN DESCRIPTION:
Elm 01 14 9.0
END DESCRIPTION:
XS GIS Cut Line= 3
      1558554.98      6810438.02      1559309.21      6809597.17
      1559842.57      6808565.99
#Sta/Elev= 30
  3727.5 1876.66  3812.4 1871.74  3890.1 1870.22  3989.5 1864.31  4038.9 1863.55
  4060.6 1861.24  4145.0 1858.41  4216.0 1857.85  4364.8 1850.98  4476.1 1849.95
  4486.3 1849.73  4740.1 1847.94  4934.9 1849.37  4980.0 1846.48  4993.1 1849.22
  4995.5 1846.48  4996.0 1845.98  5004.5 1846.48  5009.6 1849.05  5081.7 1848.00
  5208.9 1849.59  5463.3 1849.35  5557.5 1847.75  5574.0 1848.91  5596.2 1847.23
  5640.5 1849.42  5824.3 1849.62  5888.1 1851.28  5932.2 1851.18  6018.0 1852.83
#Mann=7,-1,0
  3727.5    0.07       0  4476.1   0.035       0  4486.3    0.07       0
  4995.5    0.07       0  5004.5    0.07       0  5888.1   0.035       0
  5932.2    0.07       0
Bank Sta=4995.5,5004.5
Exp/Cntr=0.3,0.1

Type RM Length L Ch R = 1,30755,515,515,515
BEGIN DESCRIPTION:
Elm 01 14 8.0
END DESCRIPTION:
XS GIS Cut Line= 3
      1559355.01      6810737.99      1559785.08      6809755.35
      1560128.18      6808667.50
#Sta/Elev= 30
  4052.3 1864.15  4061.2 1864.97  4082.5 1861.78  4136.9 1857.39  4235.9 1852.74
  4259.3 1853.52  4270.6 1851.24  4336.7 1848.22  4415.9 1845.90  4718.4 1845.21
  4969.2 1847.41  4992.0 1844.15  4995.5 1842.52  4996.0 1842.02  5004.6 1842.52
  5010.0 1843.96  5015.4 1842.82  5023.8 1844.15  5033.3 1842.52  5045.6 1846.67
  5056.5 1846.96  5195.6 1846.04  5216.5 1844.78  5241.9 1846.19  5338.9 1845.43
  5363.3 1847.10  5872.3 1847.42  6039.3 1848.78  6160.2 1851.58  6265.6 1851.74
#Mann=5,-1,0
  4052.3    0.07       0  4082.5   0.035       0  4336.7    0.07       0
  4995.5    0.07       0  5004.6    0.07       0
Bank Sta=4995.5,5004.6
Exp/Cntr=0.3,0.1

Type RM Length L Ch R = 1,30240,637,637,637
BEGIN DESCRIPTION:
Elm 01 14 7.0
END DESCRIPTION:
XS GIS Cut Line= 4
      1559455.04      6810887.97      1560083.95      6810467.39
      1560240.18      6809768.59      1560557.60      6808725.45
#Sta/Elev= 30
  3677.2 1864.02  3734.5 1860.68  3885.9 1850.23  3912.2 1849.50  4024.0 1844.29
  4282.2 1843.59  4503.6 1844.49  4545.9 1843.67  4600.6 1845.07  4627.8 1843.57
  4904.5 1845.02  4925.0 1846.08  4968.4 1844.25  4986.5 1845.17  4995.4 1842.69
  4995.9 1842.19  5004.6 1842.69  5006.7 1845.52  5027.5 1845.76  5171.4 1845.37
  5192.3 1844.08  5275.9 1844.65  5307.2 1843.06  5349.1 1845.04  5392.9 1843.85
  5420.5 1845.00  5425.7 1844.06  5458.6 1845.02  5529.5 1844.20  6240.2 1848.76
#Mann=5,-1,0
  3677.2    0.07       0  3734.5   0.035       0  3912.2    0.07       0
  4995.4    0.07       0  5004.6    0.07       0
Bank Sta=4995.4,5004.6
Exp/Cntr=0.3,0.1

Type RM Length L Ch R = 1,29603,683,683,683
BEGIN DESCRIPTION:
Elm 01 14 6.5
END DESCRIPTION:
XS GIS Cut Line= 5
      1559498.69      6810921.35      1560163.06      6810551.77
      1560662.90      6810485.19      1560895.52      6809931.19
      1560745.31      6808682.56
#Sta/Elev= 30
  4041.8 1861.78  4104.5 1858.45  4181.5 1852.87  4288.0 1847.89  4438.1 1843.78
  4985.6 1843.75  4995.4 1839.09  4995.9 1838.59  5004.7 1839.09  5005.8 1845.19
  5018.4 1844.04  5066.3 1843.52  5076.4 1844.55  5086.5 1843.63  5136.9 1842.94
  5297.2 1841.78  5355.4 1842.30  5605.1 1843.67  5683.0 1842.79  5911.3 1841.80
  5930.5 1840.39  5980.9 1841.83  6011.1 1839.97  6036.7 1842.38  6111.8 1842.11
  6152.1 1840.86  6182.3 1842.28  6414.0 1843.50  6917.6 1843.60  7164.8 1845.16
#Mann=9,-1,0
  4041.8    0.07       0  4104.5   0.035       0  4288.0    0.07       0
  4995.4    0.07       0  5004.7    0.07       0  5018.4   0.035       0
  5297.2    0.07       0  5355.4   0.035       0  5683.0    0.07       0
Bank Sta=4995.4,5004.7
Exp/Cntr=0.3,0.1

Type RM Length L Ch R = 1,28920,514,514,514
BEGIN DESCRIPTION:
Elm 01 14 6.0
END DESCRIPTION:
XS GIS Cut Line= 3
      1559607.74      6811169.50      1560837.57      6811079.94
      1561047.01      6810455.19
#Sta/Elev= 30
  4015.7 1860.14  4113.2 1856.85  4143.3 1856.96  4163.3 1854.96  4263.6 1850.28
  4331.1 1848.46  4464.1 1843.87  4518.8 1843.74  4584.5 1841.74  4664.7 1841.38
  4724.8 1840.08  4845.2 1840.60  4885.3 1840.35  4895.3 1839.72  4930.8 1840.74
  4955.4 1839.37  4965.5 1840.42  4995.5 1840.79  4998.0 1836.65  4998.3 1836.15
  5001.8 1836.15  5002.0 1836.65  5005.6 1840.72  5107.6 1840.09  5145.9 1840.51
  5186.1 1839.79  5461.8 1839.10  5540.2 1840.35  5571.8 1839.94  5907.7 1840.85
#Mann=5,-1,0
  4015.7    0.07       0  4331.1   0.035       0  4998.0   0.035       0
  5002.0   0.035       0  5107.6    0.07       0
Bank Sta=4998,5002
Exp/Cntr=0.3,0.1

Type RM Length L Ch R = 1,28406,452,452,452
BEGIN DESCRIPTION:
Elm 01 14 5.0
END DESCRIPTION:
XS GIS Cut Line= 3
      1559805.01      6811438.00      1560846.40      6811665.75
      1561111.31      6811320.97
#Sta/Elev= 30
  4241.8 1855.79  4272.5 1854.28  4315.3 1853.86  4374.9 1850.54  4436.3 1850.17
  4487.5 1847.23  4538.6 1847.20  4600.1 1843.92  4651.2 1843.79  4671.7 1842.46
  4815.0 1839.81  4970.5 1838.53  4989.0 1837.31  4998.0 1834.59  4998.3 1834.09
  5002.0 1834.59  5009.2 1836.97  5019.8 1838.11  5081.2 1838.01  5142.6 1835.68
  5163.1 1835.68  5200.1 1837.92  5225.9 1837.83  5278.5 1837.04  5307.8 1838.02
  5327.0 1836.89  5362.3 1837.38  5373.6 1836.55  5415.8 1836.57  5742.6 1837.81
#Mann=7,-1,0
  4241.8    0.07       0  4998.0    0.07       0  5002.0    0.07       0
  5225.9   0.035       0  5278.5    0.07       0  5373.6   0.035       0
  5415.8    0.07       0
Bank Sta=4998,5002
Exp/Cntr=0.3,0.1

Type RM Length L Ch R = 1,27954,438,438,438
BEGIN DESCRIPTION:
Elm 01 14 4.0
END DESCRIPTION:
XS GIS Cut Line= 3
      1559632.88      6811832.46      1560907.89      6812151.33
      1561216.25      6811823.15
#Sta/Elev= 30
  4149.3 1857.96  4203.0 1854.19  4236.5 1854.13  4277.7 1850.25  4313.8 1850.01
  4337.0 1847.33  4360.2 1846.43  4442.6 1843.95  4519.9 1843.33  4584.4 1840.99
  4664.8 1840.51  4708.1 1838.61  4915.7 1837.88  4996.7 1837.90  4998.0 1833.44
  4998.3 1832.94  5002.0 1833.44  5007.0 1838.12  5074.3 1838.20  5097.1 1838.78
  5184.7 1834.23  5220.8 1836.31  5233.8 1835.39  5343.1 1835.30  5378.1 1834.26
  5398.8 1834.95  5409.1 1833.44  5432.0 1835.15  5520.6 1834.25  5913.9 1835.49
#Mann=9,-1,0
  4149.3    0.07       0  4664.8   0.035       0  4915.7    0.07       0
  4998.0    0.07       0  5002.0    0.07       0  5074.3   0.035       0
  5220.8    0.07       0  5343.1   0.035       0  5520.6    0.07       0
Bank Sta=4998,5002
Exp/Cntr=0.3,0.1

Type RM Length L Ch R = 1,27516,478,478,478
BEGIN DESCRIPTION:
Elm 01 14 3.0
END DESCRIPTION:
XS GIS Cut Line= 3
      1559349.91      6812481.33      1561350.05      6812461.21
      1561498.77      6812066.54
#Sta/Elev= 30
  3953.1 1858.51  4138.2 1857.79  4217.0 1852.59  4278.2 1850.73  4318.2 1847.25
  4368.2 1845.58  4438.2 1841.68  4458.2 1842.18  4468.2 1841.03  4518.2 1840.17
  4558.2 1837.83  4588.2 1837.86  4628.2 1836.25  4678.2 1835.61  4788.2 1836.85
  4881.1 1836.50  4988.2 1836.02  4998.0 1831.58  4998.3 1831.08  5002.0 1831.58
  5008.2 1835.84  5058.6 1835.73  5212.3 1834.37  5408.3 1832.95  5428.3 1831.58
  5458.3 1832.71  5658.3 1831.91  5718.3 1832.85  6074.3 1832.80  6375.1 1834.11
#Mann=7,-1,0
  3953.1    0.07       0  4217.0   0.035       0  4881.1    0.07       0
  4998.0    0.07       0  5002.0    0.07       0  5058.6   0.035       0
  5212.3    0.07       0
Bank Sta=4998,5002
Exp/Cntr=0.3,0.1
