--- Elm 01 24.prj (project) ---

Proj Title=Elm 01 24 Base Level Engineering
Current Plan=p01
Default Exp/Contr=0.3,0.1
English Units
Geom File=g01
Flow File=f01
Plan File=p01
Y Axis Title=Elevation
X Axis Title(PF)=Main Channel Distance
X Axis Title(XS)=Station
BEGIN DESCRIPTION:
Elm 01 24
END DESCRIPTION:
DSS Export Rating Curves= 0
DSS Export Rating Curve Sorted= 0
DSS Export Volume Flow Curves= 0
DXF OffsetX= 0
DXF OffsetY= 0
DXF ScaleX= 1
DXF ScaleY= 10

--- Elm 01 24.p01 (plan) ---

Plan Title=Multiple Run
Program Version=4.10
Short Identifier=Multiple
Geom File=g01
Flow File=f01
Subcritical Flow
K Sum by GR= 0
Std Step Tol= 0.01
Critical Tol= 0.01
Num of Std Step Trials= 20
Max Error Tol= 0.3
Flow Tol Ratio= 0.001
Split Flow NTrial= 30
Split Flow Tol= 0.02
Split Flow Ratio= 0.02
Log Output Level= 0
Friction Slope Method= 1
Unsteady Friction Slope Method= 2
Unsteady Bridges Friction Slope Method= 1
Parabolic Critical Depth
Global Vel Dist= 1 , 1 , 1
Global Log Level= 0
CheckData=True
Encroach Param=-1 ,0,0, 0
BEGIN DESCRIPTION:
Multiple Run
END DESCRIPTION:
Computation Interval=1HOUR
Output Interval=1HOUR
Run HTab= 0
Run UNet= 0
Run PostProcess= 0
Run WQNet= 0
UNET Theta= 1
UNET Theta Warmup= 1
UNET ZTol= 0.02
UNET ZSATol= 0.05
UNET MxIter= 20
UNET MaxInSteps= 0
UNET DtIC= 0
UNET DtMin= 0
UNET MaxCRTS= 20
UNET WFStab= 2
UNET SFStab= 1
UNET WFX= 1
UNET SFX= 1
UNET DSS MLevel= 4
UNET DZMax Abort= 100
UNET Convert EG Bridges= 0
UNET Use Existing IB Tables=-1
UNET Froude Reduction=False
UNET Froude Limit= 1
UNET Froude Power= 10
UNET Time Slicing=0,0, 5
UNET Junction Losses=0
Instantaneous Interval=1HOUR
Write IC File= 0
Write IC File at Sim End=0
Echo Input=False
Echo Parameters=False
Echo Output=False
Write Detailed= 0
WQ AD Non Conservative
WQ ULTIMATE=-1
WQ Max Comp Step=1HOUR
WQ Output Interval=15MIN
WQ Output Selected Increments= 0
WQ Output face flow=0
WQ Output face velocity=0
WQ Output face area=0
WQ Output face dispersion=0
WQ Output cell volume=0
WQ Output cell surface area=0
WQ Output cell continuity=0
WQ Output cumulative cell continuity=0
WQ Output face conc=0
WQ Output face dconc_dx=0
WQ Output face courant=0
WQ Output face peclet=0
WQ Output face adv mass=0
WQ Output face disp mass=0
WQ Output cell mass=0
WQ Output cell source sink temp=0
WQ Output cell source sink nsm=0
WQ Output MaxMinRange=-1
WQ Daily Max Min Mean=-1
WQ Daily Range=0
WQ Daily Time=0
WQ Create Restart=0
WQ Fixed Restart=0
WQ System Summary=0
WQ Use Fixed Temperature=0
Sorting and Armoring Iterations= 10
XS Update Threshold= 0.02
Hydraulics Update Threshold= 0.02
Energy Slope Method= 1
Volume Change Method= 0
XS Weighting Method= 0
Number of US Weighted Cross Sections= 1
Number of DS Weighted Cross Sections= 1
Upstream XS Weight=0.25
Main XS Weight=0.5
Downstream XS Weight=0.25
Number of DS XS's Weighted with US Boundary= 1
Upstream Boundary Weight= 1
Weight of XSs Associated with US Boundary= 0
Number of US XS's Weighted with DS Boundary= 1
Downstream Boundary Weight= 0.5
Weight of XSs Associated with DS Boundary= 0.5
Sediment Output Level= 4
Mass or Volume Output= 0
Output Increment Type= 1
Profile and TS Output Increment= 10
XS Output Flag= 0
XS Output Increment= 10
Disregard all LS=0
Disregard all Conn=0
Disregard all Breaches=0
Disregard all Pumps=0

--- Elm 01 24.f01 (steady flow) ---

Flow Title=Multiple
Number of Profiles=7
Profile Names=10-year,25-year,50-year,1pct_min,100-year,1pct_plu,500-year
River Rch & RM= Elm 01 24,Reach-1,19841
     424     622     796     633    1010    1400    1670
River Rch & RM= Elm 01 24,Reach-1,19727
     540     792    1010     804    1290    1770    2110
River Rch & RM= Elm 01 24,Reach-1,13457
     630     922    1180     927    1490    2040    2410
River Rch & RM= Elm 01 24,Reach-1,6050
     717    1050    1340    1060    1690    2330    2750
Boundary for River Rch & Prof#=Elm 01 24,Reach-1,1
Up Type=0
Dn Type=3
Dn Slope=0.015
Boundary for River Rch & Prof#=Elm 01 24,Reach-1,2
Up Type=0
Dn Type=3
Dn Slope=0.015
Boundary for River Rch & Prof#=Elm 01 24,Reach-1,3
Up Type=0
Dn Type=3
Dn Slope=0.015
Boundary for River Rch & Prof#=Elm 01 24,Reach-1,4
Up Type=0
Dn Type=3
Dn Slope=0.015
Boundary for River Rch & Prof#=Elm 01 24,Reach-1,5
Up Type=0
Dn Type=3
Dn Slope=0.015
Boundary for River Rch & Prof#=Elm 01 24,Reach-1,6
Up Type=0
Dn Type=3
Dn Slope=0.015
Boundary for River Rch & Prof#=Elm 01 24,Reach-1,7
Up Type=0
Dn Type=3
Dn Slope=0.015

--- Elm 01 24.g01 (geometry) ---

Geom Title=Existing Conditions
Program Version=4.10

River Reach=Elm 01 24       ,Reach-1
Reach XY= 30
        1535805.        6802638.      1535491.56      6803501.65
      1535108.12      6803489.16      1535255.47      6803767.84
       1535054.5      6804913.04      1535304.86      6805106.34
      1535312.71       6806141.7      1535646.83      6806040.46
      1535803.78       6806598.5      1535609.77      6807882.39
      1535841.37      6808325.04      1536304.45      6808548.64
      1536054.58        6809213.      1536247.52      6809491.58
      1536007.46      6809729.83      1536244.31      6809887.46
      1536599.41      6809642.73      1536556.62      6810031.96
      1536944.76      6810627.26      1537149.98      6810492.93
      1537265.85      6810997.48      1537901.92      6811039.68
      1537612.07      6811238.01      1537904.98      6811408.19
      1537755.24      6812372.78      1538147.79      6812787.66
      1537694.49      6813747.81       1537054.6      6814167.86
      1537108.74      6814736.44        1537555.        6815238.

Type RM Length L Ch R = 1 ,19841   ,114,114,114
BEGIN DESCRIPTION:
Elm 01 24 19840.89
END DESCRIPTION:
XS GIS Cut Line= 3
      1535476.89      6802457.26      1535711.26      6802780.17
       1535914.3      6803063.04
#Sta/Elev= 30
  4597.6 1997.04  4601.2 1996.94  4633.2 1996.01  4674.9 1996.59  4733.7 1994.59
  4739.9 1992.64  4754.5 1993.03  4760.7 1991.68  4775.4  1992.2  4790.1 1991.01
  4796.3 1992.11  4804.8 1991.19    4811 1992.54    4829 1992.78  4869.7 1990.61
  4919.8 1990.61    4947 1986.27  4961.7 1986.67  4976.4 1985.56  4982.6 1986.42
  5003.8 1985.38  5004.1 1984.88  5007.8 1985.38  5183.9 1994.46  5227.8 1998.23
  5234.2 1996.84    5249 1996.23  5255.1 1997.88  5290.7 2001.79  5344.8    2006
#Mann= 5 ,-1 , 0
  4597.6    .035       0  4601.2    .063       0    4829    .035       0
  5003.8    .035       0  5007.8    .035       0
Bank Sta=5003.8,5007.8
XS Rating Curve= 0 ,0
Exp/Cntr=0.3,0.1

Type RM Length L Ch R = 1 ,19727   ,87,87,87
BEGIN DESCRIPTION:
Elm 01 24 19726.67
END DESCRIPTION:
XS GIS Cut Line= 3
      1535417.85      6802587.46      1535702.58      6802899.96
      1535910.71      6803132.18
#Sta/Elev= 30
  4585.6 1996.61    4697 1992.52  4838.9 1990.68  4845.7 1989.59  4853.1 1990.31
  4867.3 1990.04    4924 1985.45  4959.2 1985.53  4978.1  1983.5  4978.4    1983
  4982.1  1983.5  4987.5 1983.62  4994.3 1985.08  5001.7 1985.01  5093.7 1991.75
  5107.9 1993.29  5136.3 1998.97  5164.7 1994.78  5178.9 1994.35  5185.7 1995.18
  5228.3 1996.37    5235 1999.39  5242.5 1999.49  5249.2  2001.2  5263.4 2002.45
  5270.9 2002.24  5277.6 2003.36  5285.1 2002.32  5291.8 2003.25  5320.2 2002.93
#Mann= 3 ,-1 , 0
  4585.6    .035       0  4978.1    .035       0  4982.1    .035       0
Bank Sta=4978.1,4982.1
XS Rating Curve= 0 ,0
Exp/Cntr=0.3,0.1

Type RM Length L Ch R = 1 ,19640   ,129,129,129
BEGIN DESCRIPTION:
Elm 01 24 19640.25
END DESCRIPTION:
XS GIS Cut Line= 3
       1535383.1      6802698.54      1535640.08      6802958.99
      1535865.76      6803169.05
#Sta/Elev= 30
  4639.1 1996.57  4661.3 1997.38  4755.6 1993.41  4809.7 1992.51    4831 1990.12
  4859.3 1989.69  4873.4 1988.16  4894.6 1987.85  4901.7 1986.63  4944.2 1984.25
  4972.4 1984.58  4984.6 1983.12  4984.8 1982.62  4988.6 1983.12  5000.7 1985.12
  5057.2 1989.37  5112.2 1990.91  5134.9 1992.57  5142.2 1994.93  5163.2 1996.64
  5170.6 1994.63  5184.7 1993.99  5234.1 1993.61  5248.3 1995.83  5262.4 1994.88
  5276.6 1995.28  5283.9 1996.65  5290.8 1996.71  5298.1 1998.54  5313.3 1999.24
#Mann= 5 ,-1 , 0
  4639.1    .035       0  4755.6    .045       0  4984.6    .045       0
  4988.6    .045       0  5112.2    .035       0
Bank Sta=4984.6,4988.6
XS Rating Curve= 0 ,0
Exp/Cntr=0.3,0.1

Type RM Length L Ch R = 1 ,19511   ,153,153,153
BEGIN DESCRIPTION:
Elm 01 24 19511.22
END DESCRIPTION:
XS GIS Cut Line= 3
      1535273.75      6802811.42       1535530.7      6803018.02
      1535821.15      6803197.82
#Sta/Elev= 30
  4674.9 1996.84  4675.6 1996.85  4702.2 1996.66  4733.5    1995  4816.1  1993.6
    4837 1992.14  4880.1 1991.27  4894.5 1989.22  4929.7 1987.97  4985.8 1984.03
  5009.3 1983.34  5012.8  1982.4  5013.1  1981.9  5016.6  1981.9  5016.8  1982.4
  5030.2 1983.59  5072.7 1983.26  5088.1 1985.25  5103.5 1984.85  5115.5  1986.3
    5139 1986.71    5146  1987.9  5151.9 1987.33  5188.5 1988.19  5240.5 1990.87
  5286.2  1992.3  5327.2 1992.94  5335.1 1994.17    5341 1993.54  5346.2 1995.18
#Mann= 6 ,-1 , 0
  4674.9    .045       0  4675.6    .035       0  4733.5    .045       0
  5012.8    .045       0  5016.8    .045       0  5286.2    .035       0
Bank Sta=5012.8,5016.8
XS Rating Curve= 0 ,0
Exp/Cntr=0.3,0.1

Type RM Length L Ch R = 1 ,19358   ,79,79,79
BEGIN DESCRIPTION:
Elm 01 24 19358.23
END DESCRIPTION:
XS GIS Cut Line= 3
      1535225.11      6802969.38      1535542.85      6803146.49
      1535824.14      6803221.15
#Sta/Elev= 30
  4635.1 1994.39  4750.2 1994.32  4787.9 1991.42  4841.1 1990.67  4869.1 1989.32
  4875.4 1987.72  4906.8 1985.49  4912.5 1985.73  4921.2 1984.38  4944.1 1983.46
  4950.2 1982.56  4971.9 1983.34  4978.4 1982.79  4993.7 1983.04  4997.2 1982.03
  5009.4  1981.2  5009.7  1980.7  5013.2  1980.7  5013.4  1981.2  5025.6 1983.37
  5065.8 1984.13  5073.5 1985.17  5083.9 1985.25  5143.5 1988.97    5176 1990.16
  5181.2 1989.89  5216.2 1991.97  5221.3 1991.72  5270.1 1993.52  5289.9 1995.04
#Mann= 4 ,-1 , 0
  4635.1    .045       0  5009.4    .045       0  5013.4    .045       0
  5143.5    .035       0
Bank Sta=5009.4,5013.4
XS Rating Curve= 0 ,0
Exp/Cntr=0.3,0.1

Type RM Length L Ch R = 1 ,19279   ,150,150,150
BEGIN DESCRIPTION:
Elm 01 24 19278.7
END DESCRIPTION:
XS GIS Cut Line= 3
      1535195.61       6803118.7      1535508.13       6803214.2
      1535836.27      6803236.77
#Sta/Elev= 30
  4676.3  1990.9  4729.2 1989.81  4822.1 1988.83  4827.6 1989.12  4874.3 1988.03
  4884.8 1986.56  4893.2 1985.81  4898.4 1985.86  4916.2 1983.66    4926 1983.53
  4931.2 1982.53  4947.5 1981.38  4989.4  1981.6  4994.7  1980.5    4995    1980
  4998.5    1980  4998.8  1980.5    5020 1982.78    5030 1982.75    5040 1984.01
  5050.1 1984.55  5070.1 1983.43  5080.1 1983.46  5110.2 1985.41  5133.3 1986.21
  5150.3 1987.98  5176.8 1989.34  5240.5 1990.96  5276.3 1993.08    5332 1995.29
#Mann= 4 ,-1 , 0
  4676.3    .045       0  4994.7    .045       0  4998.8    .045       0
  5176.8    .035       0
Bank Sta=4994.7,4998.8
XS Rating Curve= 0 ,0
Exp/Cntr=0.3,0.1

Type RM Length L Ch R = 1 ,19129   ,143,143,143
BEGIN DESCRIPTION:
Elm 01 24 19128.71
END DESCRIPTION:
XS GIS Cut Line= 3
       1535176.5      6803192.27      1535555.01      6803347.88
      1535891.79      6803372.06
#Sta/Elev= 30
  4592.1 1989.25  4655.4 1987.83  4720.2 1988.06    4731  1987.5  4773.5 1987.64
  4808.3 1986.28  4817.5 1986.88  4832.2 1986.73  4856.2 1984.85  4861.6 1985.65
  4880.2 1983.35  4885.6 1984.76    4904 1982.95  4909.5 1981.48  4925.7 1981.66
  4933.5 1980.22  4938.9 1981.17  4947.3 1980.01  4960.8 1979.74  4961.1 1979.24
  4964.6 1979.24  4964.9 1979.74  5003.9  1981.7  5021.4 1983.15  5031.4 1983.21
  5074.7 1986.44  5081.5 1987.88  5124.4 1988.64  5171.8 1990.72    5339 1995.04
#Mann= 4 ,-1 , 0
  4592.1    .045       0  4960.8    .045       0  4964.9    .045       0
  5124.4    .035       0
Bank Sta=4960.8,4964.9
XS Rating Curve= 0 ,0
Exp/Cntr=0.3,0.1

Type RM Length L Ch R = 1 ,18986   ,82,82,82
BEGIN DESCRIPTION:
Elm 01 24 18986.31
END DESCRIPTION:
XS GIS Cut Line= 4
      1535148.78      6803197.46      1535483.83      6803424.27
      1535546.72      6803581.51      1535725.31      6803563.95
#Sta/Elev= 30
  4541.6 1989.35  4676.1 1986.66    4763 1986.79  4790.6 1985.07  4849.9 1984.05
  4855.9 1985.67  4870.9  1985.4  4876.9 1987.48  4885.8 1988.13  4891.8 1987.35
  4899.3 1987.83  4921.8 1987.04  4927.8 1985.77  4935.5  1986.5  4942.8 1985.85
  4982.5 1986.65  4988.8 1986.04  4994.2 1984.06  5013.1 1979.62  5016.4 1977.72
  5016.6 1977.22  5020.5 1977.72  5025.6 1978.95  5042.7 1980.12  5048.1 1982.53
  5062.1 1983.12  5101.9 1984.96  5169.3 1985.37  5184.8 1986.02    5295 1988.56
#Mann= 6 ,-1 , 0
  4541.6    .045       0  5016.4     .07       0  5020.5    .045       0
  5062.1     .07       0  5169.3    .045       0  5184.8     .07       0
Bank Sta=5016.4,5020.5
XS Rating Curve= 0 ,0
Exp/Cntr=0.3,0.1

Type RM Length L Ch R = 1 ,18904   ,239,239,239
BEGIN DESCRIPTION:
Elm 01 24 18871.11
END DESCRIPTION:
XS GIS Cut Line= 5
       1535108.4      6803187.85      1535296.33      6803393.02
      1535488.59       6803567.3      1535613.95      6803613.87
       1535745.4      6803644.82
#Sta/Elev= 30
  4536.3 1989.27    4622 1987.11    4693 1986.66  4735.5 1984.83  4742.3 1985.42
  4799.4 1984.47  4806.2 1986.04  4813.6 1985.28  4820.4 1987.11  4827.8 1987.31
  4834.6 1986.91  4848.8 1982.87  4869.7  1978.5  4877.2 1975.87  4891.3 1974.35
  4940.7 1974.31  4954.9  1974.5  4962.3 1975.95  4983.3 1981.97  4997.4 1983.21
  5018.4  1977.4  5023.6 1974.31  5023.9 1973.81  5027.7 1974.31  5032.6 1978.95
  5077.2 1984.69    5124 1984.01  5162.5 1984.55  5179.4 1985.98  5342.8 1988.24
#Mann= 4 ,-1 , 0
  4536.3    .045       0  4877.2     .04       0  4962.3     .07       0
  5027.7     .07       0
#XS Ineff= 2 , 0
       0  4997.4    1984               0
Permanent Ineff=
       F       F
Bank Sta=5023.6,5027.7
XS Rating Curve= 0 ,0
Exp/Cntr=0.3,0.1

Type RM Length L Ch R = 1 ,18665   ,111,111,111
BEGIN DESCRIPTION:
Elm 01 24 12.0
END DESCRIPTION:
XS GIS Cut Line= 5
      1534990.41      6803103.52      1535189.82      6803342.24
      1535252.49      6803570.26      1535404.61      6803720.79
      1535718.16      6803796.52
#Sta/Elev= 30
  4539.7 1990.81  4640.3 1989.07  4783.4 1987.05  4837.1 1986.25  4862.4 1984.37
  4898.2 1981.85  4930.7 1981.54  4939.7 1979.75  4965.1 1979.39  5002.7 1976.56
  5002.9 1976.06  5006.8 1976.56  5018.5 1977.01    5033 1978.07  5039.2 1979.98
  5044.3 1978.34  5073.6 1985.17  5078.8 1984.06  5094.5 1986.66  5158.1 1986.38
  5165.2 1985.16  5172.3 1986.61  5179.3 1984.77  5186.4 1986.35  5191.9 1983.94
  5200.6 1984.31  5207.6 1982.09  5271.3 1980.79  5383.9 1980.55  5623.8 1986.78
#Mann= 8 ,-1 , 0
  4539.7    .045       0  4640.3    .035       0  4783.4    .045       0
  4862.4     .16       0  5002.7     .07       0  5006.8     .16       0
  5018.5    .045       0  5191.9    .035       0
Bank Sta=5002.7,5006.8
XS Rating Curve= 0 ,0
Exp/Cntr=0.3,0.1

Type RM Length L Ch R = 1 ,18554   ,30,30,30
BEGIN DESCRIPTION:
Elm 01 24 18554.38
END DESCRIPTION:
XS GIS Cut Line= 5
      1534956.05      6803149.97      1535140.08       6803464.2
      1535292.85      6803620.45      1535399.52      6803724.49
       1535706.9      6803797.89
#Sta/Elev= 30
  4644.8 1991.36  4698.3 1989.24  4832.2 1987.15  4839.5 1986.57  4847.9    1983
  4868.5 1984.54  4949.5 1983.35  4999.7  1978.3    5000  1977.8  5003.8  1978.3
  5008.2 1980.51  5029.2 1984.16  5036.3 1983.52  5043.3 1985.63  5050.5  1984.1
  5057.5  1985.7  5064.6  1984.5  5095.9  1985.6  5213.1 1986.63  5227.5 1986.06
  5234.3 1983.81  5255.6 1984.77  5260.6 1982.08  5262.6 1981.01  5269.7 1983.24
  5276.7 1980.65    5298 1982.51  5361.6 1980.56  5464.4 1980.57  5692.5 1986.37
#Mann= 7 ,-1 , 0
  4644.8    .045       0  4698.3    .035       0  4868.5     .16       0
  4999.7     .07       0  5003.8     .16       0  5095.9    .045       0
  5260.6    .035       0
Bank Sta=4999.7,5003.8
XS Rating Curve= 0 ,0
Exp/Cntr=0.3,0.1

Type RM Length L Ch R = 1 ,18524   ,345,345,345
BEGIN DESCRIPTION:
Elm 01 24 10.0
END DESCRIPTION:
XS GIS Cut Line= 5
      1534866.58      6803387.73      1535099.99      6803464.73
      1535338.35      6803686.56      1535396.65      6803740.27
      1535666.79      6803798.42
#Sta/Elev= 30
  4732.6 1989.96  4855.1 1987.71  4898.5 1984.79  4958.4 1982.78  4970.4 1979.25
  5002.8 1977.18  5003.2 1976.68  5008.2 1977.18  5019.6 1979.58  5088.6 1983.53
  5104.6 1985.49  5118.8 1984.89  5125.6 1982.13    5133 1984.77  5139.8 1981.17
  5147.2 1984.48    5154 1981.49  5175.5 1983.11  5182.3 1980.38  5189.7 1983.57
  5196.5 1977.99  5210.7 1983.48  5217.5 1979.43  5224.8 1981.36  5231.7 1978.04
  5239.9  1979.5  5245.8 1977.72  5316.7 1982.12  5483.9 1980.62  5659.6 1985.06
#Mann= 8 ,-1 , 0
  4732.6    .035       0  4855.1     .16       0  4898.5     .07       0
  4958.4     .16       0  5002.8     .07       0  5008.2     .16       0
  5088.6    .045       0  5239.9    .035       0
Bank Sta=5002.8,5008.2
XS Rating Curve= 0 ,0
Exp/Cntr=0.3,0.1

Type RM Length L Ch R = 1 ,18179   ,139,139,139
BEGIN DESCRIPTION:
Elm 01 24 18299.45
END DESCRIPTION:
XS GIS Cut Line= 3
      1534815.47      6803564.92      1535126.34      6803747.51
      1535650.47      6803837.31
#Sta/Elev= 30
  4508.8 1987.62  4546.7 1986.77  4599.5  1986.8  4679.6 1985.29  4751.8 1985.61
  4759.6  1985.4  4765.4 1983.83    4793 1982.73    4833 1981.85  4845.5 1980.77
  4878.1  1980.7  4897.6 1978.06  4902.7 1978.96  4908.6 1977.06  4927.2 1976.33
    4939 1976.39  4957.6 1975.04  4969.4 1975.28    4987 1974.06  4987.5 1973.56
    4992 1973.56  4992.4 1974.06  5017.7 1978.29  5022.7 1978.18  5040.4 1980.61
  5051.1 1981.15  5080.3 1980.76  5101.3 1979.84  5212.9 1979.93  5401.1 1984.41
#Mann= 7 ,-1 , 0
  4508.8    .035       0    4793     .07       0  4927.2    .035       0
    4987    .035       0  4992.4    .035       0  5051.1     .07       0
  5080.3    .035       0
Bank Sta=4987,4992.4
XS Rating Curve= 0 ,0
Exp/Cntr=0.3,0.1

Type RM Length L Ch R = 1 ,18040   ,158,158,158
BEGIN DESCRIPTION:
Elm 01 24 18039.91
END DESCRIPTION:
XS GIS Cut Line= 3
       1534888.3      6803792.31      1535171.33      6803875.66
      1535561.95      6803953.78
#Sta/Elev= 30
  4707.3 1983.61    4756 1982.99  4872.2 1979.54  4891.7 1977.79  4919.8 1978.21
  4925.1  1977.7  4943.6 1979.26  4953.2 1978.98  4958.4 1978.44  4964.5 1976.82
  4974.9 1972.95  4982.6 1972.76  4983.1 1972.26  4987.6 1972.26    4988 1972.76
  4991.7 1974.09  5016.3 1975.24  5023.7 1974.78  5040.8 1974.73  5057.1 1975.57
  5077.5 1977.28  5097.2 1979.82  5108.1 1980.15  5128.5 1979.38  5142.8 1980.62
  5169.3 1978.88  5198.9 1978.63  5295.7 1978.63  5346.7 1979.51  5400.7 1981.55
#Mann= 7 ,-1 , 0
  4707.3    .035       0  4872.2     .07       0  4982.6     .07       0
    4988     .07       0  5023.7    .035       0  5097.2     .07       0
  5198.9    .035       0
Bank Sta=4982.6,4988
XS Rating Curve= 0 ,0
Exp/Cntr=0.3,0.1

Type RM Length L Ch R = 1 ,17882   ,42,42,42
BEGIN DESCRIPTION:
Elm 01 24 8.0
END DESCRIPTION:
XS GIS Cut Line= 3
      1534779.61      6803961.44      1535059.63      6804028.67
      1535438.73      6804032.91
#Sta/Elev= 30
  4617.5 1981.79  4643.6 1981.27  4746.4 1981.07  4799.3 1979.71  4841.2 1979.32
  4859.6 1979.74  4871.9  1980.8  4878.1 1982.38  4883.2 1982.53  4900.5 1979.46
  4905.5 1979.46  4910.8 1977.76  4940.8 1973.15  4990.9 1968.11  5008.2 1966.97
  5008.6 1966.47  5013.1 1966.47  5013.6 1966.97  5030.9  1968.1  5049.1 1971.56
    5062 1974.59  5080.9 1978.73  5090.9 1979.55  5120.9 1977.67  5140.9 1978.59
  5160.9 1977.75  5180.9 1978.12  5236.7  1977.6  5276.5 1978.12  5284.6 1978.16
#Mann= 8 ,-1 , 0
  4617.5    .035       0  4871.9     .07       0  5008.2     .07       0
  5013.6     .07       0  5049.1    .035       0    5062     .07       0
  5236.7    .035       0  5276.5     .07       0
Bank Sta=5008.2,5013.6
XS Rating Curve= 0 ,0
Exp/Cntr=0.3,0.1

Type RM Length L Ch R = 1 ,17840   ,48,48,48
BEGIN DESCRIPTION:
Elm 01 24 7.0
END DESCRIPTION:
XS GIS Cut Line= 3
      1534784.16      6804003.24      1535064.14      6804070.47
      1535441.67      6804074.69
#Sta/Elev= 30
  4622.2 1981.16  4674.5 1981.04  4695.1 1980.57  4703.5 1980.88  4777.3 1979.98
  4808.2 1979.07  4867.5 1979.48  4876.6 1980.25  4881.7 1978.55  4890.5 1977.15
  4900.7 1976.76    4908 1975.53  4913.1 1975.53  4928.3 1974.08  4928.8 1973.58
  4933.3 1973.58  4933.7 1974.08    4951 1976.96    4961 1977.54    5001 1978.18
    5031 1980.12    5041 1980.41    5061 1980.36    5071 1977.98    5081 1976.39
    5121 1977.14    5131 1978.05    5151 1976.95  5215.5 1977.53  5287.7 1977.86
#Mann= 5 ,-1 , 0
  4622.2    .035       0  4867.5     .07       0  4928.3     .07       0
  4933.7     .07       0  5215.5    .035       0
Bank Sta=4928.3,4933.7
XS Rating Curve= 0 ,0
Exp/Cntr=0.3,0.1

Type RM Length L Ch R = 1 ,17792   ,237,237,237
BEGIN DESCRIPTION:
Elm 01 24 17710.91
END DESCRIPTION:
XS GIS Cut Line= 3
      1534786.65      6804045.05      1535099.16      6804107.56
      1535470.38      6804187.35
#Sta/Elev= 30
  4625.4 1980.66  4654.3 1980.82  4764.6  1979.7  4769.7 1979.24  4820.7 1978.58
  4848.1 1979.29  4862.7 1978.61  4888.9 1977.55  4922.7 1973.76  4929.7 1972.56
  4944.1 1972.48  4950.1 1973.85  4980.8 1973.21    4991 1973.48  5001.2 1972.54
  5008.7 1970.28  5009.1 1969.78  5013.7 1969.78  5014.1 1970.28  5017.1 1971.49
  5042.1 1973.13  5052.4 1973.41  5072.8 1975.11    5083 1974.78  5094.3 1975.29
  5110.7  1975.9  5115.8 1975.73    5124 1976.85  5144.4 1976.18  5323.8 1977.25
#Mann= 5 ,-1 , 0
  4625.4    .035       0  4862.7     .07       0  5008.7     .07       0
  5014.1     .07       0  5094.3    .035       0
Bank Sta=5008.7,5014.1
XS Rating Curve= 0 ,0
Exp/Cntr=0.3,0.1

Type RM Length L Ch R = 1 ,17555   ,269,269,269
BEGIN DESCRIPTION:
Elm 01 24 17454.77
END DESCRIPTION:
XS GIS Cut Line= 3
      1534761.07      6804252.65      1535054.52      6804332.52
      1535469.43       6804403.7
#Sta/Elev= 30
  4645.7 1979.07  4720.2 1978.25  4784.5 1976.93  4815.6  1976.9    4835 1977.85
  4839.5  1977.7  4846.7 1976.59  4867.4 1975.43    4874 1974.68  4888.1 1974.06
  4929.6 1970.81  4960.5 1970.13  4980.8 1970.16  4988.2 1968.32  4988.6 1967.82
  4993.2 1967.82  4993.6 1968.32    5001 1968.55    5009 1970.17  5031.5 1970.51
  5041.6 1972.07  5051.7  1972.6  5082.2 1973.42  5112.6 1973.17    5129 1973.88
  5143.1 1973.21  5173.5 1973.35  5224.3 1974.65  5335.9 1974.69  5370.8 1973.75
#Mann= 5 ,-1 , 0
  4645.7    .035       0    4835     .07       0  4988.2     .07       0
  4993.6     .07       0  5051.7    .035       0
Bank Sta=4988.2,4993.6
XS Rating Curve= 0 ,0
Exp/Cntr=0.3,0.1

Type RM Length L Ch R = 1 ,17286   ,158,158,158
BEGIN DESCRIPTION:
Elm 01 24 17285.8
END DESCRIPTION:
XS GIS Cut Line= 3
      1534754.67      6804518.02      1535056.74      6804594.41
       1535784.2      6804782.24
#Sta/Elev= 30
  4689.1 1976.99  4761.6 1975.57  4789.2 1976.12  4802.9 1975.56  4823.5 1975.69
  4844.2 1974.61  4871.3 1974.42  4895.7 1973.46  4912.3 1972.08  4958.5 1970.89
  4978.3 1969.94  5006.5 1967.18  5006.9 1966.68  5011.5 1966.68    5012 1967.18
  5019.5 1968.28  5029.9 1968.77  5050.5 1968.47  5091.8 1968.93  5111.2 1969.64
  5116.4 1969.36  5143.5 1970.79    5157 1970.34  5164.1 1971.11  5184.8 1971.26
  5215.8 1972.24  5238.3 1971.57  5298.4 1971.19  5732.2 1970.26    5752 1970.56
#Mann= 3 ,-1 , 0
  4689.1    .035       0  5006.5    .035       0    5012    .035       0
Bank Sta=5006.5,5012
XS Rating Curve= 0 ,0
Exp/Cntr=0.3,0.1

Type RM Length L Ch R = 1 ,17128   ,195,195,195
BEGIN DESCRIPTION:
Elm 01 24 17127.89
END DESCRIPTION:
XS GIS Cut Line= 3
      1534730.39      6804672.54      1535107.09      6804736.77
      1535724.31      6804870.12
#Sta/Elev= 30
  4619.7 1976.05  4766.4  1974.4  4776.5 1973.69  4817.1 1973.01    4878 1972.89
  4916.7 1969.18  4976.9 1966.76    4982 1967.37  4998.2  1965.4  5007.2 1965.35
  5007.6 1964.85  5012.2 1964.85  5012.7 1965.35  5020.2 1965.42  5028.3 1966.57
  5033.4 1965.74  5050.9 1967.79  5071.3  1968.5  5077.6  1969.3    5102 1969.78
  5240.7 1969.47  5341.3 1969.71  5415.7 1969.22    5442 1969.49  5500.4 1969.35
  5505.5  1968.7  5531.7 1968.55  5549.6 1969.26  5554.8 1968.36  5633.3 1968.24
#Mann= 7 ,-1 , 0
  4619.7     .07       0  5007.2     .07       0  5012.7     .07       0
  5240.7    .035       0  5341.3     .07       0  5415.7    .035       0
    5442     .07       0
Bank Sta=5007.2,5012.7
XS Rating Curve= 0 ,0
Exp/Cntr=0.3,0.1

Type RM Length L Ch R = 1 ,16933   ,156,156,156
BEGIN DESCRIPTION:
Elm 01 24 16933.69
END DESCRIPTION:
XS GIS Cut Line= 3
      1534778.99      6804922.53       1535049.8      6804915.59
       1535560.5       6804915.2
#Sta/Elev= 30
    4724 1975.99    4740 1976.43    4780 1976.27  4860.1 1974.53  4900.1 1972.35
  4920.1 1972.23  4930.1 1971.26  4940.1 1970.87  4950.1 1969.07  4970.1 1967.27
  4980.1  1966.9    4990 1965.85  4994.9 1965.85  5010.1 1962.09  5017.4    1962
  5017.8  1961.5  5022.5  1961.5  5022.9    1962  5040.1 1965.04  5050.1 1965.48
  5080.1 1965.04  5120.1 1965.26  5230.1 1967.83  5330.1 1968.52  5370.1 1968.42
    5381 1968.95  5450.1 1968.29  5460.1  1968.7    5480 1967.98  5505.6  1967.7
#Mann= 5 ,-1 , 0
    4724     .07       0  5017.4     .07       0  5022.9     .07       0
    5381    .035       0    5480     .07       0
Bank Sta=5017.4,5022.9
XS Rating Curve= 0 ,0
Exp/Cntr=0.3,0.1

Type RM Length L Ch R = 1 ,16777   ,255,255,255
BEGIN DESCRIPTION:
Elm 01 24 16777.38
END DESCRIPTION:
XS GIS Cut Line= 3
      1534869.28      6805212.44      1535150.49      6805033.64
      1535445.18      6804958.32
#Sta/Elev= 30
    4666 1972.41  4676.7 1972.49  4723.5 1972.48  4775.1 1971.56  4781.1 1971.78
  4790.4 1971.24  4817.5  1971.6  4826.8 1971.06  4832.7 1971.13  4838.7 1969.68
  4862.4 1965.67  4869.1 1965.01  4905.6 1964.75  4926.7  1965.1  4984.3 1965.07
  4992.7 1964.66  4996.2 1960.87  4996.6 1960.37  5001.3 1960.37  5001.8 1960.87
  5014.2 1966.05  5041.1 1964.12    5082 1963.59  5122.8 1964.67  5148.4 1965.76
  5163.6 1967.02  5201.2 1967.42  5245.3 1967.55  5279.3 1968.26  5303.4 1968.32
#Mann= 6 ,-1 , 0
    4666    .035       0  4676.7     .07       0  4996.2     .07       0
  5001.8     .07       0  5201.2    .035       0  5279.3     .07       0
Bank Sta=4996.2,5001.8
XS Rating Curve= 0 ,0
Exp/Cntr=0.3,0.1

Type RM Length L Ch R = 1 ,16522   ,146,146,146
BEGIN DESCRIPTION:
Elm 01 24 16526.85
END DESCRIPTION:
XS GIS Cut Line= 3
      1534949.11      6805273.22      1535200.84      6805203.78
      1535410.69      6805150.29
#Sta/Elev= 30
  4631.3 1971.14  4720.4 1969.19  4740.5  1969.9  4772.3 1968.65  4785.2 1966.47
  4803.4 1965.63  4819.6 1965.99  4824.7  1965.5  4853.9 1965.99  4859.1  1965.7
  4865.6  1966.1    4876 1965.68    4892 1963.97  4917.4  1962.7  4927.7 1962.33
  4934.5 1962.69  4939.6 1961.56  4958.6 1961.86    4969 1960.39  4972.5 1959.12
    4973 1958.62  4977.7 1958.62  4978.1 1959.12  4999.9 1959.49  5010.2 1960.26
  5016.2 1960.94  5021.4 1962.84  5041.2 1962.76  5057.1 1964.01    5109 1966.08
#Mann= 3 ,-1 , 0
  4631.3     .07       0  4972.5     .07       0  4978.1     .07       0
Bank Sta=4972.5,4978.1
XS Rating Curve= 0 ,0
Exp/Cntr=0.3,0.1

Type RM Length L Ch R = 1 ,16376   ,151,151,151
BEGIN DESCRIPTION:
Elm 01 24 16375.92
END DESCRIPTION:
XS GIS Cut Line= 3
      1534924.84       6805320.1      1535310.22      6805323.57
      1535406.54      6805313.92
#Sta/Elev= 30
  4621.1 1970.84  4625.6 1970.83  4651.3 1970.66  4661.3 1970.22  4721.3 1968.72
  4761.3 1968.02  4771.3 1967.58  4781.3 1967.99  4791.3 1967.46  4821.3  1966.5
  4841.3 1966.27  4851.3  1965.3  4861.3 1964.83  4891.3 1962.23  4911.3 1961.05
  4931.3 1960.93  4944.6 1961.13  4961.3 1961.74  4971.3 1960.93  4978.5 1957.41
  4978.9 1956.91  4983.6 1956.91  4984.1 1957.41  4991.3 1959.29  5006.4 1961.46
  5014.3 1961.45  5021.3 1961.97  5071.6 1964.16  5081.6 1964.09  5103.3 1964.66
#Mann= 4 ,-1 , 0
  4621.1    .035       0  4625.6     .07       0  4978.5     .07       0
  4984.1     .07       0
Bank Sta=4978.5,4984.1
XS Rating Curve= 0 ,0
Exp/Cntr=0.3,0.1

Type RM Length L Ch R = 1 ,16225   ,181,181,181
BEGIN DESCRIPTION:
Elm 01 24 16225.17
END DESCRIPTION:
XS GIS Cut Line= 3
       1534895.3      6805467.67      1535209.52      6805439.89
       1535405.8      6805410.53
#Sta/Elev= 30
  4681.4  1970.4  4691.1 1970.04  4701.2  1970.1  4801.6 1968.34  4873.7 1966.61
  4891.9 1966.55    4912 1965.75  4932.1 1965.68  4942.1 1965.09  4952.1 1965.16
  4959.4 1964.42  4964.4 1964.85  4972.2 1963.52  4982.3 1962.52  4992.1 1960.89
  4996.8 1960.89  5012.5 1958.13  5019.8 1956.29  5020.3 1955.79    5025 1955.79
  5025.4 1956.29  5040.6 1960.73  5045.7 1959.48  5052.9 1960.67    5065 1960.43
  5084.3 1960.21  5103.5 1959.32  5114.8 1959.67  5154.1 1962.09  5195.3 1963.85
#Mann= 6 ,-1 , 0
  4681.4    .035       0  4873.7     .07       0  5019.8     .07       0
  5025.4     .07       0    5065     .16       0  5084.3     .07       0
Bank Sta=5019.8,5025.4
XS Rating Curve= 0 ,0
Exp/Cntr=0.3,0.1

Type RM Length L Ch R = 1 ,16044   ,148,148,148
BEGIN DESCRIPTION:
Elm 01 24 16044.25
END DESCRIPTION:
XS GIS Cut Line= 3
      1534938.67       6805570.1      1535355.35      6805540.59
      1535415.45      6805537.62
#Sta/Elev= 30
  4586.9 1968.88  4653.4 1967.51  4663.4 1967.03    4688 1966.79  4763.7 1965.21
  4773.7 1965.38  4783.7 1964.83  4803.8 1964.62  4811.9 1964.17  4823.8 1964.29
  4828.9 1964.76  4833.9 1964.62    4885 1961.92    4914 1959.79  4924.1 1959.71
  4934.1 1958.96  4954.1  1958.8  4964.2 1957.91  4969.8 1956.49    4972 1954.12
  4972.5 1953.62  4977.2 1953.62  4977.6 1954.12  4984.2 1954.69  4994.2  1956.9
  5001.9 1958.12    5007 1958.12  5024.3 1960.03  5035.2 1962.03  5064.8 1962.42
#Mann= 6 ,-1 , 0
  4586.9    .035       0  4811.9     .07       0    4885     .16       0
    4972     .07       0  4977.6     .16       0  5035.2    .035       0
Bank Sta=4972,4977.6
XS Rating Curve= 0 ,0
Exp/Cntr=0.3,0.1

Type RM Length L Ch R = 1 ,15896   ,199,199,199
BEGIN DESCRIPTION:
Elm 01 24 15895.67
END DESCRIPTION:
XS GIS Cut Line= 3
      1534926.57      6805698.57      1535362.09      6805688.09
      1535431.69      6805683.56
#Sta/Elev= 30
  4576.2  1968.2  4654.7 1967.01  4704.7 1965.89  4714.7 1965.32  4744.7 1964.75
  4803.7 1964.35  4814.7 1963.81  4824.7 1964.28  4844.7 1963.55  4857.2  1962.2
  4864.7 1961.23  4874.7 1960.47  4894.7 1959.59  4914.7 1959.16  4924.7 1958.18
  4934.7 1958.36  4964.7 1957.04  4984.8  1957.1  4994.8 1956.56    5002 1953.46
  5002.4 1952.96  5007.1 1952.96  5007.6 1953.46  5010.8 1956.35  5013.6 1956.35
  5024.8 1957.28  5034.8 1957.25  5064.9 1960.06  5074.9 1960.74  5081.6 1960.64
#Mann= 5 ,-1 , 0
  4576.2    .035       0  4857.2     .16       0    5002     .07       0
  5007.6     .16       0  5013.6     .07       0
Bank Sta=5002,5007.6
XS Rating Curve= 0 ,0
Exp/Cntr=0.3,0.1

Type RM Length L Ch R = 1 ,15697   ,183,183,183
BEGIN DESCRIPTION:
Elm 01 24 15697.14
END DESCRIPTION:
XS GIS Cut Line= 3
       1534925.5      6805835.29      1535214.08      6805833.12
      1535417.92      6805793.19
#Sta/Elev= 30
  4710.3 1966.85  4809.8 1965.98  4889.8 1964.33  4909.8 1964.36  4919.8 1965.29
  4939.8 1963.11  4949.8 1959.59  4959.8 1954.95    4967 1952.93  4967.5 1952.43
  4972.2 1952.43  4972.6 1952.93  4975.2 1953.43  4979.8 1954.31  4989.8 1954.08
  4996.8 1955.09  5002.2 1954.72  5020.2 1955.31  5040.6 1955.27    5061 1956.06
  5081.3  1955.6  5105.2 1955.59  5111.9 1954.94  5122.1 1955.74  5132.3 1955.83
  5142.5 1956.88  5162.9 1957.19  5180.7 1958.08  5193.4 1959.16  5206.6 1959.15
#Mann= 5 ,-1 , 0
  4710.3    .035       0    4967     .07       0  4972.6    .035       0
  4975.2     .16       0  5180.7     .07       0
Bank Sta=4967,4972.6
XS Rating Curve= 0 ,0
Exp/Cntr=0.3,0.1

Type RM Length L Ch R = 1 ,15514   ,89,89,89
BEGIN DESCRIPTION:
Elm 01 24 15514.39
END DESCRIPTION:
XS GIS Cut Line= 3
      1535003.54      6806019.76      1535307.39      6805980.69
      1535509.08      6805877.95
#Sta/Elev= 30
  4691.6 1964.46  4753.6 1963.98  4773.7 1965.17  4826.1 1962.24  4834.2 1959.26
  4841.3 1957.81  4844.3  1957.2  4854.4 1952.99  4864.5  1951.2  4874.6 1952.49
  4884.6 1951.89  4900.6 1952.75  4905.6 1951.44    4925 1951.92    4935 1954.08
  4945.1 1955.22  4965.3 1954.68  4985.5 1953.02  4994.2 1951.13    4998 1951.13
  5003.7 1949.04  5004.1 1948.54  5009.3 1949.04  5019.1 1949.27  5041.4  1954.2
    5058 1952.91  5096.3 1953.91  5118.7 1955.54  5129.3 1957.17  5224.3  1957.6
#Mann= 5 ,-1 , 0
  4691.6    .035       0  4841.3     .16       0  5003.7     .07       0
  5009.3     .16       0  5129.3     .07       0
Bank Sta=5003.7,5009.3
XS Rating Curve= 0 ,0
Exp/Cntr=0.3,0.1

Type RM Length L Ch R = 1 ,15425   ,136,136,136
BEGIN DESCRIPTION:
Elm 01 24 15424.57
END DESCRIPTION:
XS GIS Cut Line= 3
      1535031.77      6806082.69      1535355.14      6806054.48
      1535591.49      6805874.46
#Sta/Elev= 30
  4676.5 1963.35  4709.9 1964.72  4756.7 1962.96  4870.5 1959.62  4890.5 1958.39
  4899.3 1957.04  4904.3 1957.25  4920.7 1955.31  5001.1 1950.31  5005.4 1948.82
  5010.7 1948.72  5011.1 1948.22  5015.8 1948.22  5016.3 1948.72  5019.9 1950.53
  5034.4 1952.46    5049 1952.07  5098.9 1952.58  5110.2 1953.29  5148.8 1954.29
  5155.1 1955.02  5163.3 1955.01  5169.6 1956.08  5190.4 1956.13  5198.7 1955.18
  5219.5 1956.66    5234 1954.91  5263.1 1954.62  5269.4 1955.85  5298.2 1955.64
#Mann= 5 ,-1 , 0
  4676.5    .035       0  4756.7     .16       0  5010.7     .07       0
  5016.3     .16       0  5110.2     .07       0
Bank Sta=5010.7,5016.3
XS Rating Curve= 0 ,0
Exp/Cntr=0.3,0.1

Type RM Length L Ch R = 1 ,15289   ,389,389,389
BEGIN DESCRIPTION:
Elm 01 24 15288.56
END DESCRIPTION:
XS GIS Cut Line= 3
      1535170.72      6806251.94      1535337.78      6806167.32
      1535795.71      6805754.96
#Sta/Elev= 30
  4815.7 1961.87  4875.3  1963.3  4897.6 1962.23  4903.2 1959.97  4910.2 1959.24
  4925.5 1959.31  4942.2 1957.06  4947.8 1957.39  4964.4  1952.8    4970 1954.18
  4977.4 1949.88  4983.9 1947.42  4984.4 1946.92  4989.5 1947.42  4992.3 1947.57
  5007.7 1950.17  5071.2 1951.69  5167.2 1950.19  5234.2 1952.16  5248.4 1951.48
  5255.1 1952.46  5276.8 1951.21  5283.5 1952.35    5291 1951.79  5354.5 1953.71
  5389.6 1956.17  5411.3 1955.35  5499.8 1955.82  5545.9 1955.46  5619.2 1956.76
#Mann= 7 ,-1 , 0
  4815.7     .07       0  4983.9     .07       0  4989.5     .07       0
  4992.3     .16       0  5167.2     .07       0  5499.8    .035       0
  5545.9     .07       0
Bank Sta=4983.9,4989.5
XS Rating Curve= 0 ,0
Exp/Cntr=0.3,0.1

Type RM Length L Ch R = 1 ,14900   ,151,151,151
BEGIN DESCRIPTION:
Elm 01 24 14900.38
END DESCRIPTION:
XS GIS Cut Line= 3
      1535300.88      6806334.43      1535602.53      6806104.39
      1535836.88       6805794.1
#Sta/Elev= 30
  4543.4 1959.03    4623 1957.15  4658.3 1957.28  4732.6 1954.41  4758.1 1953.29
  4785.8 1949.93    4808  1948.3  4850.4 1948.71  4965.2 1947.96    4986 1947.27
  4990.6 1945.71  4991.1 1945.21  4995.8 1945.21  4996.2 1945.71  5000.6 1948.03
  5006.9 1948.33  5015.2 1951.58  5021.4 1951.15    5036 1953.68  5050.6 1952.67
  5057.5  1953.8  5071.4 1955.11  5079.7 1954.86  5085.9 1956.05  5089.7 1955.74
  5100.5 1954.53  5106.8 1954.97  5151.8 1954.36  5235.8 1954.64  5311.6 1956.81
#Mann= 8 ,-1 , 0
  4543.4     .07       0  4732.6     .16       0  4785.8     .07       0
  4990.6     .07       0  4996.2     .07       0  5057.5    .035       0
  5089.7     .07       0  5151.8    .035       0
Bank Sta=4990.6,4996.2
XS Rating Curve= 0 ,0
Exp/Cntr=0.3,0.1

Type RM Length L Ch R = 1 ,14749   ,233,233,233
BEGIN DESCRIPTION:
Elm 01 24 14748.66
END DESCRIPTION:
XS GIS Cut Line= 3
      1535355.12      6806343.11      1535693.68      6806180.34
      1536041.56      6805985.88
#Sta/Elev= 30
  4622.9 1957.98    4671 1957.47  4678.2 1958.48  4700.4 1955.41  4755.9 1955.48
  4761.5 1954.29  4778.1 1953.15  4784.2  1950.4  4789.7 1950.84  4800.3 1947.46
  4806.8  1946.6  4920.6 1947.36  4993.6 1945.83  4994.1 1945.33  4999.4 1945.83
  5037.1 1947.18  5080.5    1950  5090.8 1949.79  5103.2 1951.36  5112.5 1950.78
  5118.2 1951.83  5126.1 1950.73  5134.2 1950.87    5149 1951.58  5155.9 1953.07
  5171.9 1952.25  5193.6 1953.07  5199.3 1954.47  5248.9 1953.58  5397.1  1955.4
#Mann= 5 ,-1 , 0
  4622.9     .07       0  4920.6    .035       0  4993.6    .035       0
  4999.4    .035       0  5248.9     .07       0
Bank Sta=4993.6,4999.4
XS Rating Curve= 0 ,0
Exp/Cntr=0.3,0.1

Type RM Length L Ch R = 1 ,14516   ,226,226,226
BEGIN DESCRIPTION:
Elm 01 24 14515.95
END DESCRIPTION:
XS GIS Cut Line= 3
      1535352.93       6806401.7      1535752.27        6806380.
      1536140.36      6806293.27
#Sta/Elev= 30
  4597.9 1958.56    4620 1958.33    4640 1957.09  4660.1 1957.35  4720.2 1954.71
  4730.2 1955.15  4780.2 1953.68  4820.3 1951.14  4850.3 1947.15  4870.4 1945.52
    4939  1944.8  4960.5 1945.85  4970.5    1945  4977.6    1943  4978.1  1942.5
    4983  1942.5  4983.4    1943  4990.6 1944.93  4996.7 1945.46  5028.1 1945.17
  5033.2  1945.7  5062.1 1944.14  5076.6 1944.49  5103.1 1948.02  5162.8 1950.55
  5225.8 1951.29  5236.3 1951.44  5246.5 1950.39  5330.4 1951.32  5395.5 1951.68
#Mann= 6 ,-1 , 0
  4597.9     .07       0  4977.6     .07       0  4983.4     .07       0
  5162.8    .035       0  5225.8     .07       0  5330.4    .035       0
Bank Sta=4977.6,4983.4
XS Rating Curve= 0 ,0
Exp/Cntr=0.3,0.1

Type RM Length L Ch R = 1 ,14290   ,203,203,203
BEGIN DESCRIPTION:
Elm 01 24 14290.06
END DESCRIPTION:
XS GIS Cut Line= 3
      1535435.47      6806601.35      1535800.02       6806590.5
       1536177.6      6806477.66
#Sta/Elev= 30
  4634.4 1954.09  4663.9 1953.93    4674 1953.45    4694 1951.34    4704 1951.71
  4743.9 1949.95    4754 1949.83  4784.9 1947.19    4814 1944.61  4821.1 1942.58
  4821.6 1942.08  4826.5 1942.08  4826.9 1942.58    4844 1942.61    4864 1943.53
  4934.1 1944.27  5027.9 1943.76  5040.2 1943.28  5055.8 1943.85    5061  1943.1
  5066.9  1943.2  5087.8 1945.12  5094.1 1944.99  5119.1  1946.4  5132.4  1946.5
    5140  1945.6  5160.3 1945.56  5246.2 1948.33  5252.9 1948.64  5393.2 1950.06
#Mann= 8 ,-1 , 0
  4634.4     .07       0  4743.9     .16       0  4784.9     .07       0
  4821.1     .07       0  4826.9     .07       0  5040.2    .035       0
  5246.2     .07       0  5252.9    .035       0
Bank Sta=4821.1,4826.9
XS Rating Curve= 0 ,0
Exp/Cntr=0.3,0.1

Type RM Length L Ch R = 1 ,14087   ,303,303,303
BEGIN DESCRIPTION:
Elm 01 24 14133.8
END DESCRIPTION:
XS GIS Cut Line= 3
      1535454.72      6806715.49      1535754.06       6806798.2
       1536256.8      6806744.99
#Sta/Elev= 30
  4638.5 1947.17  4658.5 1946.69    4700 1945.77  4721.8 1947.14  4732.2 1946.93
  4739.6 1944.87  4744.8 1947.21  4752.9 1944.84  4763.3 1943.75  4784.3 1943.31
    4814 1941.49  4835.9 1940.43  4877.4 1940.67  4892.5 1938.64  4898.2 1940.63
    4932 1944.69  4960.1 1946.04  4970.1 1945.25  4990.2 1942.22  4996.8 1939.31
  5007.4 1938.35  5007.9 1937.85  5013.2 1938.35  5030.4 1939.75  5040.5 1942.04
  5050.6 1942.54  5094.6 1942.18    5161 1942.98  5251.7 1944.17  5454.6 1948.34
#Mann= 6 ,-1 , 0
  4638.5     .07       0  4658.5     .16       0    4814     .07       0
  5007.4     .07       0  5013.2     .07       0    5161    .035       0
Bank Sta=5007.4,5013.2
XS Rating Curve= 0 ,0
Exp/Cntr=0.3,0.1

Type RM Length L Ch R = 1 ,13784   ,327,327,327
BEGIN DESCRIPTION:
Elm 01 24 13774.35
END DESCRIPTION:
XS GIS Cut Line= 4
      1535504.86      6806766.61       1535618.4      6806988.36
      1535771.44      6807065.38      1536320.97      6807119.05
#Sta/Elev= 30
    4546 1945.89  4555.2 1945.41  4560.8 1948.59  4577.4 1945.59    4583 1947.16
  4599.6 1943.74  4637.4 1942.24  4659.9 1939.67  4671.9 1943.99  4688.5 1946.26
  4732.9  1943.8  4795.1 1944.94  4801.2 1944.57  4813.7 1940.48  4823.5  1941.2
  4829.1 1937.35  4845.8 1939.46  4851.4 1937.08  4890.5 1938.39  4957.4 1937.76
  5000.2 1936.72  5007.3 1934.55  5007.8 1934.05  5013.2 1934.55  5020.3 1937.67
  5023.5 1937.55  5045.1 1936.57  5100.7 1941.82  5146.8 1941.14  5518.6 1946.75
#Mann= 4 ,-1 , 0
    4546     .16       0  5007.3     .07       0  5013.2     .16       0
  5023.5    .035       0
Bank Sta=5007.3,5013.2
XS Rating Curve= 0 ,0
Exp/Cntr=0.3,0.1

Type RM Length L Ch R = 1 ,13457   ,187,187,187
BEGIN DESCRIPTION:
Elm 01 24 13456.54
END DESCRIPTION:
XS GIS Cut Line= 3
      1535110.18      6807338.89      1535606.61      6807234.91
      1536141.67      6807308.48
#Sta/Elev= 30
  4494.6 1942.35  4591.5 1943.48  4736.2 1942.71  4775.4 1942.65  4785.6 1943.35
    4806 1941.84  4813.6  1940.6  4818.7 1941.21  4863.5  1936.9  4877.6 1937.11
    4898 1935.62  4908.2 1935.86  4913.4 1936.88  4962.7 1934.44  4974.8 1931.28
  4975.3 1930.78  4984.7 1931.28  4989.9 1933.39  4998.4 1934.85  5020.4 1935.92
  5050.6 1935.94  5070.8 1934.86  5111.2 1935.14  5177.8  1938.1  5202.1 1938.48
  5207.6 1939.56  5222.2 1940.13  5242.4 1939.17  5284.6 1939.21  5541.9 1941.03
#Mann= 6 ,-1 , 0
  4494.6    .035       0  4736.2     .07       0  4962.7     .16       0
  4974.8     .07       0  4984.7     .16       0  5177.8    .035       0
Bank Sta=4974.8,4984.7
XS Rating Curve= 0 ,0
Exp/Cntr=0.3,0.1

Type RM Length L Ch R = 1 ,13270   ,439,439,439
BEGIN DESCRIPTION:
Elm 01 24 13270.46
END DESCRIPTION:
XS GIS Cut Line= 3
      1535063.21      6807399.26      1535593.19       6807389.2
      1536170.01      6807332.19
#Sta/Elev= 30
  4507.8 1941.87  4549.6  1941.4  4609.6 1942.05  4749.6 1941.67  4809.6 1940.62
  4819.6 1941.36  4829.6 1941.05  4836.1 1939.72  4859.6 1938.13  4869.7 1936.69
  4889.7 1935.11  4929.7 1933.56  4969.7 1934.21  4989.7 1933.68  5004.7 1931.06
  5005.2 1930.56  5014.2 1930.56  5014.7 1931.06  5019.7 1932.09  5029.7 1932.89
  5069.8  1934.2  5108.4 1933.38  5140.2  1933.7  5160.3 1934.71  5168.6 1934.42
  5208.8 1937.35  5230.6 1938.62  5270.8  1938.2  5351.2 1938.56  5617.5 1940.98
#Mann= 6 ,-1 , 0
  4507.8    .035       0  5004.7    .035       0  5014.7    .035       0
  5108.4     .07       0  5168.6     .16       0  5208.8    .035       0
Bank Sta=5004.7,5014.7
XS Rating Curve= 0 ,0
Exp/Cntr=0.3,0.1

Type RM Length L Ch R = 1 ,12831   ,240,240,240
BEGIN DESCRIPTION:
Elm 01 24 12831.04
END DESCRIPTION:
XS GIS Cut Line= 3
      1535046.43       6807637.4      1535653.57      6807613.92
      1536201.82      6807369.88
#Sta/Elev= 30
  4226.5  1943.7  4468.4  1940.7  4495.3 1941.46  4533.7 1940.16  4599.8  1936.9
  4622.1 1936.75  4675.4 1935.43  4695.4 1935.76    4740 1934.86  4814.4 1934.42
  4885.2  1932.3    4978  1932.8  4989.1 1931.94  4999.8 1932.18  5006.9 1930.79
  5007.4 1929.16  5007.9 1928.66  5016.9 1928.66  5017.4 1929.16  5021.7  1931.3
  5035.6 1933.16  5043.6 1936.03  5053.4 1937.23  5065.5 1937.72  5082.1 1936.04
  5122.3 1937.18  5142.1 1937.88  5151.8 1937.24  5273.5 1939.05  5434.2 1940.32
#Mann= 9 ,-1 , 0
  4226.5    .035       0  4468.4     .07       0  4533.7    .035       0
  4622.1     .07       0    4740    .035       0  4814.4     .07       0
  5007.4     .07       0  5017.4     .07       0  5122.3    .035       0
Bank Sta=5007.4,5017.4
XS Rating Curve= 0 ,0
Exp/Cntr=0.3,0.1

Type RM Length L Ch R = 1 ,12591   ,142,142,142
BEGIN DESCRIPTION:
Elm 01 24 12590.99
END DESCRIPTION:
XS GIS Cut Line= 3
      1534989.46      6807647.46      1535660.27      6807731.31
      1536317.66      6807684.36
#Sta/Elev= 30
  4320.2 1944.53  4529.2 1941.72  4537.4 1941.55  4547.5 1940.44  4567.7 1941.33
  4597.9 1940.38  4691.3 1939.13  4728.9 1937.89  4759.1 1938.56  4766.1 1937.45
  4779.3 1937.08  4819.6 1937.01  4890.1 1934.62  4960.7  1933.9  4980.8 1932.05
    5021 1931.28  5031.1 1930.24  5036.1 1928.91  5036.6 1928.41  5045.6 1928.41
  5046.1 1928.91  5051.1 1930.13  5061.1 1930.91  5081.2 1931.05  5151.4 1933.69
  5181.4 1933.21    5255 1934.57  5510.4 1935.74  5547.4 1936.06  5655.3 1936.16
#Mann= 6 ,-1 , 0
  4320.2    .035       0  4691.3     .07       0  5036.1     .07       0
  5046.1     .07       0  5510.4    .035       0  5547.4     .07       0
Bank Sta=5036.1,5046.1
XS Rating Curve= 0 ,0
Exp/Cntr=0.3,0.1

Type RM Length L Ch R = 1 ,12449   ,302,302,302
BEGIN DESCRIPTION:
Elm 01 24 12449.47
END DESCRIPTION:
XS GIS Cut Line= 3
      1535019.64      6807778.27      1535603.25      6807855.42
      1536314.31      6807892.31
#Sta/Elev= 30
  4408.5 1944.57  4441.9 1943.62  4504.7 1943.04  4546.9  1942.1  4585.4  1941.8
  4605.6 1940.71  4706.4 1939.63  4824.3 1937.13  4847.6 1937.05  4918.3 1934.84
  4958.6 1934.12  4981.3 1933.76  5000.6 1934.05    5009 1932.35    5014 1927.99
  5014.5 1927.49  5023.5 1927.49    5024 1927.99    5029 1930.53    5049 1930.64
    5069 1929.74  5129.1 1930.89  5143.8 1930.69  5159.2 1931.83  5269.3 1931.99
  5409.5 1934.04  5499.6 1934.14  5559.7 1934.85  5637.8 1934.55  5709.2  1934.6
#Mann= 5 ,-1 , 0
  4408.5    .035       0  4546.9     .07       0    5014     .07       0
    5024     .07       0  5637.8    .035       0
Bank Sta=5014,5024
XS Rating Curve= 0 ,0
Exp/Cntr=0.3,0.1

Type RM Length L Ch R = 1 ,12147   ,195,195,195
BEGIN DESCRIPTION:
Elm 01 24 12146.6
END DESCRIPTION:
XS GIS Cut Line= 3
      1535076.64      6807939.27       1535804.5      6808039.89
      1536378.06      6808060.02
#Sta/Elev= 30
  4264.5 1943.04  4303.2 1941.97  4433.6 1941.03  4454.7 1940.11  4545.5 1938.23
  4555.6  1937.2  4659.2 1935.64  4666.6 1934.52  4737.3 1932.63  4767.6  1932.6
  4797.9 1930.98  4908.9 1930.32  4969.5 1929.37  4979.6 1928.61  4984.6 1926.58
  4985.1 1926.08  4994.2 1926.08  4994.7 1926.58    4997 1927.12    5002 1927.12
  5009.8 1929.52  5029.8 1932.05    5067 1932.52  5139.9  1934.1  5169.9 1933.83
  5209.9 1934.45  5433.4 1934.06  5530.1  1933.7  5560.1  1934.3  5573.2  1933.5
#Mann= 5 ,-1 , 0
  4264.5    .035       0  4984.6    .035       0  4994.7    .035       0
    5067     .07       0  5433.4    .035       0
Bank Sta=4984.6,4994.7
XS Rating Curve= 0 ,0
Exp/Cntr=0.3,0.1

Type RM Length L Ch R = 1 ,11952   ,635,635,635
BEGIN DESCRIPTION:
Elm 01 24 11951.73
END DESCRIPTION:
XS GIS Cut Line= 3
       1535153.8      6808053.31      1535801.15       6808207.6
      1536305.99      6808216.28
#Sta/Elev= 30
  4332.7 1942.09  4436.7 1940.51  4498.4 1938.31    4519 1938.47  4529.3 1937.68
  4630.1  1933.9  4693.7 1932.68  4734.9 1932.51  4761.6 1930.46  4893.1 1930.16
  4899.3 1929.45  4935.3 1928.42    4961 1928.79  4971.3 1927.92  4977.5 1925.64
    4978 1925.14  4987.1 1925.14  4987.6 1925.64  4991.9 1926.09  4997.6 1928.73
    5012 1929.15    5032 1931.19    5062 1932.39    5102  1932.8  5162.1  1932.4
  5192.1 1933.31  5212.1    1933  5302.1 1933.51  5362.4  1933.1  5503.1 1933.43
#Mann= 4 ,-1 , 0
  4332.7     .07       0  4977.5     .07       0  4987.6     .07       0
  5362.4    .035       0
Bank Sta=4977.5,4987.6
XS Rating Curve= 0 ,0
Exp/Cntr=0.3,0.1

Type RM Length L Ch R = 1 ,11317   ,221,221,221
BEGIN DESCRIPTION:
Elm 01 24 11316.61
END DESCRIPTION:
XS GIS Cut Line= 3
      1535207.46      6808281.38      1536260.66      6808489.34
      1536461.82      6808488.58
#Sta/Elev= 30
  3931.1 1943.34  4122.3 1936.05  4141.7  1936.4  4152.8    1935  4244.3    1930
  4305.8 1927.49  4387.3 1928.24    4479 1926.69  4519.8 1927.57    4530 1929.27
  4540.2 1928.79  4550.4  1925.5  4565.7 1923.77  4566.2 1923.27  4575.8 1923.77
  4591.1 1924.56  4601.3 1927.43  4608.5 1927.89  4621.7 1927.41  4642.1 1924.06
  4652.3 1924.56  4659.8 1927.69  4703.3 1926.33  4805.2 1925.53  4870.1 1925.26
  4907.1  1926.3  4978.5 1925.36  5009.3 1923.92    5089 1931.18  5205.8 1930.56
#Mann= 3 ,-1 , 0
  3931.1     .07       0  4565.7     .07       0  4575.8     .07       0
Bank Sta=4565.7,4575.8
XS Rating Curve= 0 ,0
Exp/Cntr=0.3,0.1

Type RM Length L Ch R = 1 ,11096   ,181,181,181
BEGIN DESCRIPTION:
Elm 01 24 11096.41
END DESCRIPTION:
XS GIS Cut Line= 3
      1535147.07      6808475.92      1536220.41       6808660.4
       1536601.4      6808713.87
#Sta/Elev= 30
  3900.6 1945.33  3969.5  1943.8  4020.3 1940.43  4040.5 1940.59  4050.7 1938.51
  4183.1  1933.2  4352.8 1928.77  4446.4 1925.23  4477.8    1925  4532.7 1926.57
  4608.8  1926.2  4659.5 1927.03  4669.6 1924.13  4674.7 1921.32  4675.2 1920.82
  4684.8 1921.32  4700.1 1925.59  4811.7 1925.43  4827.4 1923.71  4862.4  1923.5
  4892.9 1925.31  4923.3 1925.67  4963.9 1923.79  5024.6  1924.5  5044.8  1922.3
    5065 1924.34  5085.3 1924.64  5125.6 1929.12  5156.6 1928.12  5374.4 1926.96
#Mann= 3 ,-1 , 0
  3900.6     .07       0  4674.7     .07       0  4684.8     .07       0
Bank Sta=4674.7,4684.8
XS Rating Curve= 0 ,0
Exp/Cntr=0.3,0.1

Type RM Length L Ch R = 1 ,10915   ,352,352,352
BEGIN DESCRIPTION:
Elm 01 24 10914.76
END DESCRIPTION:
XS GIS Cut Line= 3
      1535207.47      6808794.57      1536156.68      6808814.69
      1536619.51      6808858.29
#Sta/Elev= 30
    4052  1940.3  4189.6 1942.22  4269.6 1940.51  4299.6 1938.19  4319.6 1933.85
  4339.6 1928.39  4349.6 1927.15  4359.6 1926.15  4409.6 1924.68  4549.6 1924.42
  4579.6 1923.79  4689.7 1925.25  4769.7  1924.5  4799.7 1925.05  4819.7  1921.6
  4829.7 1921.35  4849.7  1924.8  4869.7 1923.32  4909.7 1921.86  4969.7 1923.01
  4979.7 1921.83  4984.7 1920.49  4985.2 1919.99  4994.3 1919.99  4994.8 1920.49
  5009.8 1922.31  5092.6 1923.25  5140.4 1925.24  5299.7 1926.73  5466.3 1926.28
#Mann= 3 ,-1 , 0
    4052     .07       0  4984.7     .07       0  4994.8     .07       0
Bank Sta=4984.7,4994.8
XS Rating Curve= 0 ,0
Exp/Cntr=0.3,0.1
