--- Elm 01 31.prj (project) ---

Proj Title=Elm 01 31 Base Level Engineering
Current Plan=p01
Default Exp/Contr=0.3,0.1
English Units
Geom File=g01
Flow File=f01
Plan File=p01
Y Axis Title=Elevation
X Axis Title(PF)=Main Channel Distance
X Axis Title(XS)=Station
BEGIN DESCRIPTION:
Elm 01 31
END DESCRIPTION:
DSS Export Rating Curves= 0
DSS Export Rating Curve Sorted= 0
DSS Export Volume Flow Curves= 0
DXF OffsetX= 0
DXF OffsetY= 0
DXF ScaleX= 1
DXF ScaleY= 10

--- Elm 01 31.p01 (plan) ---

Plan Title=Multiple Run
Program Version=4.10
Short Identifier=Multiple
Geom File=g01
Flow File=f01
Subcritical Flow
K Sum by GR= 0
Std Step Tol= 0.01
Critical Tol= 0.01
Num of Std Step Trials= 20
Max Error Tol= 0.3
Flow Tol Ratio= 0.001
Split Flow NTrial= 30
Split Flow Tol= 0.02
Split Flow Ratio= 0.02
Log Output Level= 0
Friction Slope Method= 1
Unsteady Friction Slope Method= 2
Unsteady Bridges Friction Slope Method= 1
Parabolic Critical Depth
Global Vel Dist= 1 , 1 , 1
Global Log Level= 0
CheckData=True
Encroach Param=-1 ,0,0, 0
BEGIN DESCRIPTION:
Multiple Run
END DESCRIPTION:
Computation Interval=1HOUR
Output Interval=1HOUR
Run HTab= 0
Run UNet= 0
Run PostProcess= 0
Run WQNet= 0
UNET Theta= 1
UNET Theta Warmup= 1
UNET ZTol= 0.02
UNET ZSATol= 0.05
UNET MxIter= 20
UNET MaxInSteps= 0
UNET DtIC= 0
UNET DtMin= 0
UNET MaxCRTS= 20
UNET WFStab= 2
UNET SFStab= 1
UNET WFX= 1
UNET SFX= 1
UNET DSS MLevel= 4
UNET DZMax Abort= 100
UNET Convert EG Bridges= 0
UNET Use Existing IB Tables=-1
UNET Froude Reduction=False
UNET Froude Limit= 1
UNET Froude Power= 10
UNET Time Slicing=0,0, 5
UNET Junction Losses=0
Instantaneous Interval=1HOUR
Write IC File= 0
Write IC File at Sim End=0
Echo Input=False
Echo Parameters=False
Echo Output=False
Write Detailed= 0
WQ AD Non Conservative
WQ ULTIMATE=-1
WQ Max Comp Step=1HOUR
WQ Output Interval=15MIN
WQ Output Selected Increments= 0
WQ Output face flow=0
WQ Output face velocity=0
WQ Output face area=0
WQ Output face dispersion=0
WQ Output cell volume=0
WQ Output cell surface area=0
WQ Output cell continuity=0
WQ Output cumulative cell continuity=0
WQ Output face conc=0
WQ Output face dconc_dx=0
WQ Output face courant=0
WQ Output face peclet=0
WQ Output face adv mass=0
WQ Output face disp mass=0
WQ Output cell mass=0
WQ Output cell source sink temp=0
WQ Output cell source sink nsm=0
WQ Output MaxMinRange=-1
WQ Daily Max Min Mean=-1
WQ Daily Range=0
WQ Daily Time=0
WQ Create Restart=0
WQ Fixed Restart=0
WQ System Summary=0
WQ Use Fixed Temperature=0
Sorting and Armoring Iterations= 10
XS Update Threshold= 0.02
Hydraulics Update Threshold= 0.02
Energy Slope Method= 1
Volume Change Method= 0
XS Weighting Method= 0
Number of US Weighted Cross Sections= 1
Number of DS Weighted Cross Sections= 1
Upstream XS Weight=0.25
Main XS Weight=0.5
Downstream XS Weight=0.25
Number of DS XS's Weighted with US Boundary= 1
Upstream Boundary Weight= 1
Weight of XSs Associated with US Boundary= 0
Number of US XS's Weighted with DS Boundary= 1
Downstream Boundary Weight= 0.5
Weight of XSs Associated with DS Boundary= 0.5
Sediment Output Level= 4
Mass or Volume Output= 0
Output Increment Type= 1
Profile and TS Output Increment= 10
XS Output Flag= 0
XS Output Increment= 10
Disregard all LS=0
Disregard all Conn=0
Disregard all Breaches=0
Disregard all Pumps=0

--- Elm 01 31.f01 (steady flow) ---

Flow Title=Multiple
Number of Profiles=7
Profile Names=10-year,25-year,50-year,1pct_min,100-year,1pct_plu,500-year
River Rch & RM= Elm 01 31,Reach-1,18349
     222     307     376     286     459     632     692
River Rch & RM= Elm 01 31,Reach-1,16028
     346     487     605     466     746    1030    1150
River Rch & RM= Elm 01 31,Reach-1,9334
     444     631     788     609     977    1340    1520
Boundary for River Rch & Prof#=Elm 01 31,Reach-1,1
Up Type=0
Dn Type=3
Dn Slope=0.005
Boundary for River Rch & Prof#=Elm 01 31,Reach-1,2
Up Type=0
Dn Type=3
Dn Slope=0.005
Boundary for River Rch & Prof#=Elm 01 31,Reach-1,3
Up Type=0
Dn Type=3
Dn Slope=0.005
Boundary for River Rch & Prof#=Elm 01 31,Reach-1,4
Up Type=0
Dn Type=3
Dn Slope=0.005
Boundary for River Rch & Prof#=Elm 01 31,Reach-1,5
Up Type=0
Dn Type=3
Dn Slope=0.005
Boundary for River Rch & Prof#=Elm 01 31,Reach-1,6
Up Type=0
Dn Type=3
Dn Slope=0.005
Boundary for River Rch & Prof#=Elm 01 31,Reach-1,7
Up Type=0
Dn Type=3
Dn Slope=0.005

--- Elm 01 31.g01 (geometry) ---

Geom Title=Existing Conditions
Program Version=4.10

River Reach=Elm 01 31       ,Reach-1
Reach XY= 30
        1551655.        6813088.      1551651.46      6813686.54
      1551010.28      6814035.29      1550451.17      6816236.42
      1549962.33       6817087.9      1550154.95      6817858.04
      1550060.39      6818290.44      1550239.78      6818387.76
      1550544.56      6818239.03      1550938.57      6818420.38
      1550996.96      6818641.32      1550863.96      6818844.67
      1551496.87      6819081.92      1552004.41      6820427.39
      1551563.24      6821234.76      1551099.53      6822940.45
      1550992.99      6823086.83      1550790.88      6823051.32
      1550794.68      6823298.18      1550552.69      6823293.08
      1550407.58      6823533.03      1550021.05      6823520.95
      1550154.07      6823877.52      1549849.48      6824540.43
       1549358.1      6824839.65      1549597.17      6825234.73
       1549505.2      6825722.66      1549702.37      6826029.52
      1549520.36      6826138.11        1549255.        6825988.

Type RM Length L Ch R = 1 ,18349   ,350,350,350
BEGIN DESCRIPTION:
Elm 01 31 18348.96
END DESCRIPTION:
XS GIS Cut Line= 3
      1551160.98      6813219.36      1551655.08       6813182.2
      1552055.05      6813137.99
#Sta/Elev= 30
  4504.5 1888.59  4528.6 1888.13    4669 1887.87  4699.1 1887.29  4739.2 1887.55
  4809.4 1886.76  4829.4 1887.11  4889.6 1886.28  4899.6 1886.97  4909.7 1886.91
  4919.7 1886.02  4929.7 1886.34  4969.8  1884.7  4979.9 1883.79  4987.1 1881.89
  4992.1 1881.44  4995.5 1880.26  4995.7 1879.76  4999.2 1879.76  4999.5 1880.26
  5030.1  1883.1  5040.2 1885.09  5060.3 1884.79  5138.7 1885.98  5191.1 1886.72
  5204.9 1886.27  5231.3 1886.19  5301.7 1887.59  5351.9 1889.21  5402.4 1890.03
#Mann= 5 ,-1 , 0
  4504.5     .07       0  4995.5     .07       0  4999.5     .07       0
  5138.7    .035       0  5204.9     .07       0
Bank Sta=4995.5,4999.5
XS Rating Curve= 0 ,0
Exp/Cntr=0.3,0.1

Type RM Length L Ch R = 1 ,17999   ,307,307,307
BEGIN DESCRIPTION:
Elm 01 31 17999.25
END DESCRIPTION:
XS GIS Cut Line= 2
      1551136.65      6813486.72      1552131.58      6813573.39
#Sta/Elev= 30
  4479.3 1886.27  4497.7 1886.74  4537.9 1885.96  4658.3 1885.49  4670.1 1884.79
  4728.6 1884.91  4788.8  1884.7  4818.9  1884.1  4889.2 1884.13  4919.3 1883.47
  4972.7 1881.48  4999.6 1880.66  5006.6 1879.41  5006.9 1878.91  5010.4 1878.91
  5010.6 1879.41  5013.6 1879.78  5029.7 1880.09  5039.8 1881.92  5052.9 1883.02
  5059.8 1883.57    5090 1883.86  5167.3 1883.84  5320.8 1884.81  5362.1 1885.82
  5407.7 1887.47  5451.3 1888.96  5469.9    1890    5475 1889.79    5478  1890.3
#Mann= 7 ,-1 , 0
  4479.3     .07       0  4972.7    .035       0  5006.6    .035       0
  5010.6    .035       0  5052.9     .07       0  5167.3    .035       0
  5407.7     .07       0
Bank Sta=5006.6,5010.6
XS Rating Curve= 0 ,0
Exp/Cntr=0.3,0.1

Type RM Length L Ch R = 1 ,17692   ,236,236,236
BEGIN DESCRIPTION:
Elm 01 31 17691.93
END DESCRIPTION:
XS GIS Cut Line= 3
       1551174.8      6813535.31      1551549.83      6813799.22
       1551893.6        6814268.
#Sta/Elev= 30
  4545.4 1885.27  4611.9 1884.42  4677.2 1884.52  4683.3 1883.99  4712.9 1884.27
  4727.7  1884.1  4733.8 1883.56  4855.8 1882.35  4927.2 1882.33    4942 1881.86
    4963 1879.64  4992.6 1879.78  4998.6  1877.3  5004.5 1877.11  5004.7 1876.61
  5008.2 1876.61  5008.5 1877.11  5014.9 1878.78  5027.3 1881.01    5042 1882.12
  5136.1 1880.44    5157 1880.52  5171.6 1882.04  5177.8    1882  5186.3 1882.76
  5207.1 1882.03  5236.4 1881.77  5336.8 1882.48  5499.7 1884.63  5585.3 1884.62
#Mann= 3 ,-1 , 0
  4545.4     .07       0  5004.5     .07       0  5008.5     .07       0
Bank Sta=5004.5,5008.5
XS Rating Curve= 0 ,0
Exp/Cntr=0.3,0.1

Type RM Length L Ch R = 1 ,17456   ,213,213,213
BEGIN DESCRIPTION:
Elm 01 31 17455.93
END DESCRIPTION:
XS GIS Cut Line= 3
      1550973.48      6813594.39      1551344.97      6813903.39
      1551733.84      6814288.79
#Sta/Elev= 30
  4519.1 1885.69  4707.1 1884.23  4721.5 1884.63  4742.3 1883.72  4842.5 1882.97
    4935 1882.93  4949.3 1882.65  4955.8 1881.08  4990.9 1876.76  4996.8 1876.63
    4997 1876.13  5000.8 1876.63  5012.7 1876.68  5019.7 1877.83  5026.8  1877.7
    5041 1879.12  5100.5    1880  5111.7 1880.51  5118.7 1881.97  5182.4 1881.78
  5189.4    1884  5196.1 1882.57  5203.6 1882.82  5210.7 1881.55  5224.8 1881.38
  5458.1 1881.82  5486.4 1882.48  5493.5  1881.9  5500.6 1882.73  5549.8 1883.61
#Mann= 5 ,-1 , 0
  4519.1     .07       0  4996.8     .07       0  5000.8     .07       0
  5100.5    .035       0  5196.1     .07       0
Bank Sta=4996.8,5000.8
XS Rating Curve= 0 ,0
Exp/Cntr=0.3,0.1

Type RM Length L Ch R = 1 ,17243   ,336,336,336
BEGIN DESCRIPTION:
Elm 01 31 17272.36
END DESCRIPTION:
XS GIS Cut Line= 3
      1550738.51      6813719.53      1551144.72      6813972.98
      1551568.37      6814292.45
#Sta/Elev= 30
  4506.3 1885.74    4757 1884.38    4836 1882.97  4879.3  1883.8  4924.5 1882.77
  4945.8 1880.06  4951.7 1878.03  4971.6 1875.89  4971.9 1875.39  4975.6 1875.89
    5003 1877.85  5032.1 1877.71  5046.7 1878.44  5052.9  1879.9  5067.5 1880.95
  5073.8 1882.95  5088.3 1884.35  5096.6 1884.16  5102.9 1882.63    5132 1881.41
    5182  1881.6  5202.8 1880.58  5214.8 1880.86  5296.5 1881.44  5367.3 1880.75
  5388.1 1881.23  5396.4 1882.16  5422.9 1880.94  5452.6 1881.65  5515.7 1881.47
#Mann= 5 ,-1 , 0
  4506.3     .07       0  4971.6     .07       0  4975.6     .07       0
  5214.8    .035       0  5422.9     .07       0
Bank Sta=4971.6,4975.6
XS Rating Curve= 0 ,0
Exp/Cntr=0.3,0.1

Type RM Length L Ch R = 1 ,16907   ,105,105,105
BEGIN DESCRIPTION:
Elm 01 31 17003.62
END DESCRIPTION:
XS GIS Cut Line= 3
      1550529.93      6814072.46      1550974.39      6814169.68
      1551451.79      6814311.52
#Sta/Elev= 30
  4469.1 1883.49  4475.5 1882.32  4514.3 1883.45  4519.4 1882.26  4607.1  1883.7
  4612.3 1882.14  4648.3 1883.66  4656.1  1883.5  4661.2 1882.32  4689.3 1883.53
    4749 1882.99  4754.1 1881.91  4771.2 1882.98  4803.1 1882.83  4863.3 1881.47
  4873.5 1880.14  4914.5 1877.54  4919.8 1876.08  4920.1 1875.58  4923.8 1876.08
  4971.2 1878.35  4976.9  1880.1  5042.9  1880.1  5070.8 1883.26  5102.1 1879.17
  5147.7 1880.07  5154.2 1880.94  5180.9 1880.17  5251.3 1880.74  5422.1 1881.47
#Mann= 4 ,-1 , 0
  4469.1     .07       0  4919.8     .07       0  4923.8     .07       0
  5251.3    .035       0
Bank Sta=4919.8,4923.8
XS Rating Curve= 0 ,0
Exp/Cntr=0.3,0.1

Type RM Length L Ch R = 1 ,16802   ,223,223,223
BEGIN DESCRIPTION:
Elm 01 31 16695.61
END DESCRIPTION:
XS GIS Cut Line= 3
      1550424.51      6814175.77      1550924.46       6814259.1
      1551476.52      6814356.32
#Sta/Elev= 30
  4441.6  1882.2  4634.7 1882.88  4736.1  1882.3  4766.5 1880.33  4785.7 1881.36
  4827.3 1880.43  4907.4 1880.91  4938.9 1880.08  4951.3  1879.1  4959.2 1876.83
  4972.7 1876.82  4979.5  1875.1  4987.6 1874.98  4987.9 1874.48  4991.6 1874.98
  5009.9 1875.89  5026.9 1879.37  5091.2 1879.27  5111.5 1882.15  5121.6 1881.76
  5140.4 1878.94  5172.4 1880.37  5294.2 1880.36  5313.2 1881.53  5318.3 1880.93
  5324.7 1882.07    5345 1881.09  5372.5 1881.79  5377.5 1880.79    5509 1881.85
#Mann= 3 ,-1 , 0
  4441.6    .035       0  4987.6    .035       0  4991.6    .035       0
Bank Sta=4987.6,4991.6
XS Rating Curve= 0 ,0
Exp/Cntr=0.3,0.1

Type RM Length L Ch R = 1 ,16579   ,348,348,348
BEGIN DESCRIPTION:
Elm 01 31 16455.89
END DESCRIPTION:
XS GIS Cut Line= 3
      1550395.48      6814346.31       1550871.2      6814457.43
      1551390.99      6814564.85
#Sta/Elev= 30
  4478.7    1881  4562.2 1880.56    4662  1879.7  4686.4 1880.54  4745.2 1879.93
  4786.3 1878.05  4813.9 1879.06  4837.6 1877.84  4868.4 1878.99  4919.8  1879.2
  4971.7  1876.8  4995.7 1873.69    5012 1874.36  5020.2 1873.22  5020.4 1872.72
  5024.2 1873.22  5032.4 1874.66  5045.9 1874.87  5052.8 1876.72  5083.7 1877.93
  5103.9 1878.18  5124.3 1879.72  5134.5 1879.27  5141.3 1877.32  5154.9 1876.78
  5185.5 1876.95  5191.5 1878.25  5219.2 1878.15  5318.3 1880.07    5498 1881.77
#Mann= 7 ,-1 , 0
  4478.7     .07       0  4562.2    .035       0    4662     .07       0
  5020.2     .07       0  5024.2     .07       0  5083.7    .035       0
  5219.2     .07       0
Bank Sta=5020.2,5024.2
XS Rating Curve= 0 ,0
Exp/Cntr=0.3,0.1

Type RM Length L Ch R = 1 ,16231   ,203,203,203
BEGIN DESCRIPTION:
Elm 01 31 16230.56
END DESCRIPTION:
XS GIS Cut Line= 3
       1550265.1        6814702.      1550848.44      6814795.75
      1551258.21      6814875.62
#Sta/Elev= 30
  4412.2  1879.7  4472.9 1879.71  4523.9 1878.74  4641.6 1877.11  4715.9 1875.86
  4746.3 1874.69  4794.3 1876.06  4817.2 1874.48  4861.2 1875.04  4936.4 1874.34
    4959 1872.92    4983 1870.16  4983.3 1869.66  4986.8 1869.66    4987 1870.16
  4998.7  1871.6  5009.7 1872.06  5019.9 1874.25  5030.1 1875.66    5081 1876.13
  5094.7 1877.84  5101.4 1877.44  5121.8 1874.62  5126.6 1874.53  5152.3 1874.53
  5172.7 1875.73  5249.6  1877.2  5359.2  1878.2  5409.5 1878.97  5420.5 1879.64
#Mann= 8 ,-1 , 0
  4412.2     .07       0  4523.9    .035       0  4641.6     .07       0
  4936.4    .035       0    4983    .035       0    4987    .035       0
  5126.6     .07       0  5359.2    .035       0
Bank Sta=4983,4987
XS Rating Curve= 0 ,0
Exp/Cntr=0.3,0.1

Type RM Length L Ch R = 1 ,16028   ,236,236,236
BEGIN DESCRIPTION:
Elm 01 31 16028.3
END DESCRIPTION:
XS GIS Cut Line= 3
      1550292.91      6814879.09      1550817.19      6814986.72
      1551247.76      6815049.22
#Sta/Elev= 30
  4480.4 1878.26  4524.9  1877.8  4663.4 1875.41  4737.7 1874.69  4758.2 1873.48
  4778.6 1874.82  4819.4 1873.47  4846.4  1874.2  4931.7  1874.3  4941.9 1873.97
    4955 1872.54  4990.4 1869.29  4990.7 1868.79  4994.3 1868.79  4994.6 1869.29
  5011.9  1872.6  5023.5 1873.53  5033.6 1874.02    5074 1873.86  5094.2 1876.66
  5114.5 1873.67  5128.2 1873.69  5144.8 1873.65  5194.4 1875.24  5235.7 1874.99
  5255.9  1875.8  5296.3 1875.72  5316.5 1876.73  5369.2 1877.62  5450.7 1878.29
#Mann= 8 ,-1 , 0
  4480.4     .07       0  4524.9    .035       0  4663.4     .07       0
    4955    .035       0  4990.4    .035       0  4994.6    .035       0
  5128.2     .07       0  5369.2    .035       0
Bank Sta=4990.4,4994.6
XS Rating Curve= 0 ,0
Exp/Cntr=0.3,0.1

Type RM Length L Ch R = 1 ,15792   ,200,200,200
BEGIN DESCRIPTION:
Elm 01 31 15791.88
END DESCRIPTION:
XS GIS Cut Line= 3
      1550049.78      6815045.74      1550699.13      6815188.11
      1551150.25      6815264.45
#Sta/Elev= 30
  4324.7 1877.05    4330 1876.46  4391.5 1876.27  4449.9    1877  4568.6  1875.7
  4732.7 1874.48    4760 1874.29  4790.7 1872.75    4826 1873.87  4852.2 1872.81
  4882.9 1874.11  4967.7 1873.54  4989.5 1872.04  5012.6 1868.36  5012.9 1867.86
  5016.8 1868.36  5019.8 1868.53    5036 1868.95  5046.1 1870.79  5075.1 1873.56
  5117.1 1873.63  5127.3 1874.36  5135.5 1875.98  5157.7 1872.44  5179.3 1872.36
  5218.6 1874.12  5261.3 1873.28  5316.7 1875.39  5423.8 1875.76    5447  1876.1
#Mann= 8 ,-1 , 0
  4324.7     .07       0  4568.6    .035       0  4732.7     .07       0
  5012.6     .07       0  5016.8     .07       0  5019.8    .035       0
  5179.3     .07       0  5423.8    .035       0
Bank Sta=5012.6,5016.8
XS Rating Curve= 0 ,0
Exp/Cntr=0.3,0.1

Type RM Length L Ch R = 1 ,15592   ,322,322,322
BEGIN DESCRIPTION:
Elm 01 31 15591.55
END DESCRIPTION:
XS GIS Cut Line= 3
      1550074.09      6815247.13      1550660.94      6815375.61
      1551139.47      6815483.11
#Sta/Elev= 30
  4392.5 1875.35  4403.7 1875.85  4413.9 1877.43  4424.6 1875.44    4506 1874.56
  4567.3  1874.9  4754.1 1872.93  4782.4 1871.94  4823.4 1873.71  4854.1 1871.83
  4883.6 1873.09  4956.5 1872.86  4981.5 1871.59  4992.8 1869.25  5007.7 1868.54
  5015.8 1866.35  5016.1 1865.85    5020 1866.35    5025  1868.3  5037.1 1869.42
  5068.3 1872.54  5110.1 1873.81  5121.9  1875.5  5130.6 1875.54  5151.1 1871.84
  5184.7 1871.78  5208.5 1873.09  5243.4 1871.11  5284.4 1873.48  5483.7 1874.86
#Mann= 7 ,-1 , 0
  4392.5     .07       0  4567.3    .035       0  4754.1     .07       0
  5015.8     .07       0    5020     .07       0  5037.1    .035       0
  5184.7     .07       0
Bank Sta=5015.8,5020
XS Rating Curve= 0 ,0
Exp/Cntr=0.3,0.1

Type RM Length L Ch R = 1 ,15270   ,389,389,389
BEGIN DESCRIPTION:
Elm 01 31 15270.44
END DESCRIPTION:
XS GIS Cut Line= 3
      1549959.56      6815531.86      1550601.91       6815663.8
      1551160.45      6815750.53
#Sta/Elev= 30
  4341.2 1875.69  4450.1 1875.69  4742.1 1872.97  4785.7 1869.89  4806.2  1872.3
    4848 1870.56  4928.7 1870.46  4959.3 1869.66  4994.8 1864.18  4995.1 1863.68
  4999.1 1864.18  5040.6 1868.42  5081.1 1868.63  5111.4 1874.08  5124.3 1872.89
  5131.6 1870.41  5141.8 1869.56  5182.2 1869.93  5202.5 1871.81  5222.7 1871.35
  5232.8 1869.36    5243 1869.17  5250.2 1870.86  5263.2 1872.05  5293.6 1872.87
  5386.2 1873.05  5435.2 1874.48  5455.5 1873.22  5506.1 1872.81  5562.2 1873.76
#Mann= 3 ,-1 , 0
  4341.2    .035       0  4994.8    .035       0  4999.1    .035       0
Bank Sta=4994.8,4999.1
XS Rating Curve= 0 ,0
Exp/Cntr=0.3,0.1

Type RM Length L Ch R = 1 ,14881   ,194,194,194
BEGIN DESCRIPTION:
Elm 01 31 14880.64
END DESCRIPTION:
XS GIS Cut Line= 3
      1549810.25      6815858.25      1550497.75      6816021.44
      1551100.99      6816135.85
#Sta/Elev= 30
  4285.2 1875.12  4403.1  1873.3  4479.6 1873.51  4598.6 1872.27    4738 1870.38
  4793.4 1868.02  4814.3 1869.12  4855.4 1866.81  4906.8 1867.23  4968.4 1866.34
  4991.8 1864.91    5000 1862.48  5000.3 1861.98  5004.5 1862.48  5019.5 1864.19
    5030 1864.14  5080.6 1865.51    5101 1869.89  5106.8 1872.09  5121.3 1871.05
  5141.7 1867.94  5194.6 1867.65  5211.3 1868.34  5243.5 1866.28  5263.6 1869.22
  5309.8  1870.3  5345.2  1871.2    5447 1871.81    5488  1871.2  5605.8 1872.36
#Mann= 8 ,-1 , 0
  4285.2     .07       0  4598.6    .035       0  4793.4     .07       0
    5000     .07       0  5004.5     .07       0    5030    .035       0
  5194.6     .07       0  5309.8    .035       0
Bank Sta=5000,5004.5
XS Rating Curve= 0 ,0
Exp/Cntr=0.3,0.1

Type RM Length L Ch R = 1 ,14687   ,214,214,214
BEGIN DESCRIPTION:
Elm 01 31 14687.32
END DESCRIPTION:
XS GIS Cut Line= 3
      1549744.25      6816087.41      1550463.02        6816202.
      1551140.08      6816365.19
#Sta/Elev= 30
  4279.9  1873.9  4564.7 1871.31    4706 1868.42  4776.8  1868.1  4797.1 1866.64
  4807.2 1868.12    4828  1867.9  4847.7 1863.22  4857.9 1863.31  4878.1 1866.08
  4890.2 1865.27  4918.6 1866.33  4938.9 1861.06    4967 1860.23  4967.3 1859.73
  4971.5 1860.23  5030.4  1860.5  5050.2  1865.1  5055.4 1865.18  5081.8 1870.52
  5092.1 1871.59  5102.4 1871.54  5133.2 1865.79  5192.9 1864.81  5215.5 1863.99
  5228.2 1865.39  5256.7 1865.59  5306.9 1867.76  5390.4 1869.13  5704.2 1871.11
#Mann= 5 ,-1 , 0
  4279.9     .07       0  4564.7    .035       0    4967    .035       0
  4971.5    .035       0  5192.9     .07       0
Bank Sta=4967,4971.5
XS Rating Curve= 0 ,0
Exp/Cntr=0.3,0.1

Type RM Length L Ch R = 1 ,14473   ,293,293,293
BEGIN DESCRIPTION:
Elm 01 31 14473.37
END DESCRIPTION:
XS GIS Cut Line= 3
      1549782.49      6816288.81       1550365.8      6816386.03
      1551028.96      6816521.44
#Sta/Elev= 30
    4413 1871.45  4518.6 1870.83  4702.2 1868.04  4838.3 1866.52  4912.3 1865.46
  4921.2 1865.74  4932.6 1868.55    4963 1861.84  4973.1 1860.45  4999.1 1860.31
  4999.4 1859.81  5003.7 1860.31  5044.4 1860.59  5054.6 1861.66  5084.6 1868.89
  5095.4 1869.56    5126  1862.1  5146.4 1866.37  5156.6 1866.12  5166.8 1864.59
  5185.7 1864.14  5190.8 1862.95  5217.9 1863.05  5228.1 1864.24  5258.7 1865.08
  5286.7 1864.23  5319.9 1865.74  5330.1 1864.52  5432.2 1867.51  5681.2 1869.42
#Mann= 6 ,-1 , 0
    4413    .045       0  4518.6     .07       0  4702.2    .035       0
  4838.3     .07       0  4999.1     .07       0  5003.7     .07       0
Bank Sta=4999.1,5003.7
XS Rating Curve= 0 ,0
Exp/Cntr=0.3,0.1

Type RM Length L Ch R = 1 ,14180   ,338,338,338
BEGIN DESCRIPTION:
Elm 01 31 14180.36
END DESCRIPTION:
XS GIS Cut Line= 3
      1549692.19      6816552.69      1550265.11      6816642.97
      1550878.84      6816733.12
#Sta/Elev= 30
  4435.9 1869.49  4580.9 1868.82  4698.5  1867.6  4893.5  1865.4  4904.4 1867.65
  4914.5 1868.11  4924.7 1867.58    4956 1861.86  4995.5  1860.6  5015.9 1862.97
  5025.9 1867.41    5036 1869.44  5046.1 1869.61  5066.3 1864.12  5096.6 1860.51
  5124.7 1860.33    5125 1859.83  5129.3 1860.33    5158 1864.24  5187.6 1863.78
  5217.7 1861.41  5222.7 1863.17  5238.1 1863.93  5308.9 1862.76    5319  1863.7
  5329.1 1862.12  5369.5 1861.74  5399.9 1863.64  5480.7 1865.38  5636.2 1866.76
#Mann= 6 ,-1 , 0
  4435.9    .045       0  4580.9     .07       0  4698.5    .035       0
  4893.5     .07       0  5124.7     .07       0  5129.3     .07       0
Bank Sta=5124.7,5129.3
XS Rating Curve= 0 ,0
Exp/Cntr=0.3,0.1

Type RM Length L Ch R = 1 ,13842   ,513,513,513
BEGIN DESCRIPTION:
Elm 01 31 13841.82
END DESCRIPTION:
XS GIS Cut Line= 3
      1549494.31      6816799.23       1550053.3      6816906.86
      1550824.13      6817045.75
#Sta/Elev= 30
  4427.1 1868.94  4687.1 1867.61    4715 1867.65  4855.5 1866.39  4958.4 1863.93
  4974.3  1860.8  5027.2 1860.77  5032.3 1861.07  5059.1 1868.29  5069.2  1868.2
  5079.4 1867.15  5085.9 1863.98  5099.7 1861.73  5144.6 1858.25  5188.8 1857.57
  5189.1 1857.07  5193.5 1857.57  5221.6 1859.24  5251.8 1867.41  5256.9 1865.97
  5262.3 1867.08  5282.6 1860.47  5323.2 1859.94  5343.6 1858.05  5394.4 1861.13
  5455.3 1862.42  5506.1 1860.71  5516.3 1862.44  5556.9 1860.76  5779.6 1865.08
#Mann= 6 ,-1 , 0
  4427.1    .045       0  4687.1     .07       0    4715    .035       0
  4958.4     .07       0  5188.8     .07       0  5193.5     .07       0
Bank Sta=5188.8,5193.5
XS Rating Curve= 0 ,0
Exp/Cntr=0.3,0.1

Type RM Length L Ch R = 1 ,13329   ,196,196,196
BEGIN DESCRIPTION:
Elm 01 31 13467.89
END DESCRIPTION:
XS GIS Cut Line= 3
      1549473.41      6817142.95      1549935.61      6817391.43
       1550811.6      6817145.55
#Sta/Elev= 30
    4403 1868.57  4425.3 1868.47  4481.2 1868.08  4591.9 1867.14  4796.8 1865.77
  4866.2 1866.08  4871.8 1864.69  4888.1 1865.85  4893.8 1862.14  4904.3 1865.36
    4910 1861.07  4942.7 1861.56  5001.2 1861.81  5034.6 1868.69  5041.4 1868.31
  5068.6 1858.67  5082.9 1857.13  5121.8 1856.67  5122.2 1856.17  5127.2 1856.67
  5333.2  1856.9  5401.3  1858.3  5406.5  1857.2  5435.4 1858.47  5479.9 1857.42
  5560.7 1861.41  5626.6 1860.78  5773.3 1864.31  5778.8 1862.67  5837.6 1864.47
#Mann= 9 ,-1 , 0
    4403     .07       0  4425.3    .045       0  4481.2     .07       0
  4591.9    .035       0  4796.8     .07       0  4942.7    .035       0
  5001.2     .07       0  5121.8    .035       0  5127.2     .07       0
Bank Sta=5121.8,5127.2
XS Rating Curve= 0 ,0
Exp/Cntr=0.3,0.1

Type RM Length L Ch R = 1 ,13133   ,397,397,397
BEGIN DESCRIPTION:
Elm 01 31 13133.23
END DESCRIPTION:
XS GIS Cut Line= 3
       1549383.2      6817552.69       1550053.3      6817552.69
      1550768.62      6817354.77
#Sta/Elev= 30
  4328.5  1866.5  4537.4 1865.58  4660.3  1865.9  4680.3 1864.34  4710.6 1864.09
  4930.3 1863.37  4950.3 1862.78  4960.3 1859.64  4990.5 1861.01  5010.7 1861.81
  5035.8 1866.64  5052.2 1862.41  5070.1 1861.22  5075.3 1862.37  5093.7 1860.64
  5104.1 1858.23  5109.6 1855.57  5122.2 1854.58  5122.6 1854.08  5127.6 1854.58
  5143.9 1855.61    5156 1859.43  5188.6 1859.18  5222.9 1857.28  5275.4  1857.3
  5331.1 1856.25  5456.9 1859.77  5550.3 1860.29  5597.2 1859.12  5740.8 1859.87
#Mann= 7 ,-1 , 0
  4328.5     .07       0  4537.4    .035       0  4710.6     .07       0
  4990.5    .035       0  5122.2    .035       0  5127.6    .035       0
  5275.4     .07       0
Bank Sta=5122.2,5127.6
XS Rating Curve= 0 ,0
Exp/Cntr=0.3,0.1

Type RM Length L Ch R = 1 ,12736   ,339,339,339
BEGIN DESCRIPTION:
Elm 01 31 12735.71
END DESCRIPTION:
XS GIS Cut Line= 3
      1549414.39      6817941.58      1550150.52      6817920.75
       1550775.5       6817615.2
#Sta/Elev= 30
  4259.3 1864.83  4351.2 1864.44  4516.2 1863.07  4920.7 1861.63  4990.2 1857.37
  5037.9 1863.87  5045.2 1863.15  5054.9  1859.2  5105.5 1856.17  5134.3 1852.07
    5157 1852.33    5218 1853.72  5223.6 1855.18  5240.5 1852.38  5246.1 1854.08
  5282.9 1851.16  5283.3 1850.66  5288.3 1851.16  5323.5    1852  5377.9 1860.12
  5381.2 1859.42  5390.3 1863.92  5398.1 1863.87  5420.7 1860.33  5465.7 1858.52
  5501.6 1861.46  5600.8  1857.5  5623.3 1858.07  5651.5 1861.95  5691.4 1857.92
#Mann= 8 ,-1 , 0
  4259.3     .07       0  4351.2    .035       0  4516.2     .07       0
    5157    .033       0  5282.9     .07       0  5288.3    .033       0
  5377.9     .07       0  5651.5    .035       0
Bank Sta=5282.9,5288.3
XS Rating Curve= 0 ,0
Exp/Cntr=0.3,0.1

Type RM Length L Ch R = 1 ,12397   ,197,197,197
BEGIN DESCRIPTION:
Elm 01 31 12396.89
END DESCRIPTION:
XS GIS Cut Line= 3
      1549282.46      6818472.83      1550056.77       6818226.3
      1550771.05      6817636.85
#Sta/Elev= 30
  4188.5 1863.72  4243.1 1864.15  4307.2  1863.7    4480 1862.55    4949 1859.42
  5005.8 1854.55  5026.6  1855.7  5032.5 1858.25  5038.8 1858.79  5063.1 1863.03
  5090.5 1863.05  5098.3 1859.29    5127 1856.23    5222 1853.45  5379.6 1849.86
    5380 1849.36  5385.1 1849.86    5467 1850.67    5515 1856.55  5524.3 1860.05
  5538.7 1861.44  5559.5    1861  5567.4 1857.96  5581.7 1857.05  5744.5 1857.05
  5773.2 1861.95  5808.4 1857.73  5881.2 1857.43  5915.2 1860.54  5927.2 1858.83
#Mann= 11 ,-1 , 0
  4188.5    .035       0  4243.1     .07       0  4307.2    .035       0
    4480     .07       0  5032.5     .16       0  5038.8     .07       0
    5222    .033       0  5379.6     .07       0  5385.1    .033       0
    5515     .07       0  5881.2    .035       0
Bank Sta=5379.6,5385.1
XS Rating Curve= 0 ,0
Exp/Cntr=0.3,0.1

Type RM Length L Ch R = 1 ,12200   ,460,460,460
BEGIN DESCRIPTION:
Elm 01 31 12186.87
END DESCRIPTION:
XS GIS Cut Line= 3
      1549640.11      6819011.02      1550436.16      6818038.15
      1550808.98        6817672.
#Sta/Elev= 30
  4188.5 1861.45    4251 1858.02  4418.3 1857.97  4712.6 1858.16  4784.3 1859.37
  4982.5 1857.34  4994.1 1855.15  4994.5 1854.65  4999.6 1855.15  5060.7  1856.4
  5075.1 1857.47    5083 1859.56  5089.4 1858.34  5103.8 1861.52  5178.1 1861.66
  5239.3 1861.72  5293.4 1861.35  5401.2 1861.47  5448.2 1861.15  5494.3 1855.36
  5791.4 1856.84  5805.5 1857.15  5826.7 1861.37  5850.2 1859.27  5876.2 1857.03
  5897.4 1858.26  5904.5 1857.13  5925.7 1857.81  5932.8 1856.25  5968.1 1856.66
#Mann= 9 ,-1 , 0
  4188.5    .035       0  4418.3     .07       0  4994.1     .07       0
  4999.6     .07       0  5178.1     .16       0  5239.3     .07       0
  5293.4     .16       0  5401.2     .07       0  5850.2    .035       0
Bank Sta=4994.1,4999.6
XS Rating Curve= 0 ,0
Exp/Cntr=0.3,0.1

Type RM Length L Ch R = 1 ,11740   ,472,472,472
BEGIN DESCRIPTION:
Elm 01 31 11736.79
END DESCRIPTION:
XS GIS Cut Line= 3
      1549976.74      6818975.04      1550499.58      6818336.45
      1550920.41      6817623.74
#Sta/Elev= 30
  4065.7 1856.73  4346.2 1855.32  4403.3 1858.35  4432.1 1867.73  4567.5 1868.38
  4602.9  1868.3  4609.3 1864.98  4617.2 1867.78  4623.7 1864.41  4638.1 1868.55
  4687.6 1862.31  4701.9 1866.91  4829.7 1855.22  4844.1  1859.6  4864.9 1856.09
  4872.8 1858.86  4879.2 1854.98  4891.1 1858.08  4893.4 1854.79  4967.6 1853.03
  5014.1 1847.24  5014.6 1846.74  5019.8 1847.24  5047.6 1857.87  5090.5 1860.97
  5121.8 1857.96  5170.5 1854.06  5521.7 1859.89  5628.1 1857.71  5718.7 1857.83
#Mann= 7 ,-1 , 0
  4065.7     .07       0  4567.5     .16       0  4891.1     .07       0
  5014.1     .07       0  5019.8     .07       0  5121.8    .035       0
  5628.1     .07       0
Bank Sta=5014.1,5019.8
XS Rating Curve= 0 ,0
Exp/Cntr=0.3,0.1

Type RM Length L Ch R = 1 ,11268   ,626,626,626
BEGIN DESCRIPTION:
Elm 01 31 11268.35
END DESCRIPTION:
XS GIS Cut Line= 3
      1550379.67      6819132.59      1550938.72      6818417.28
      1551289.39        6817893.
#Sta/Elev= 30
  4094.5 1856.83  4336.9 1855.46  4351.3 1856.75  4379.5 1867.44    4393 1868.96
  4415.5    1864  4450.8 1850.18  4486.1 1847.69  4497.7 1844.46  4498.2 1843.96
  4503.4 1844.46  4506.1 1844.46  4849.1 1844.46  4877.7 1853.92  4885.8 1852.94
  4899.9 1845.88  4906.6 1844.46  5013.5 1844.46  5023.2 1845.54  5042.1 1849.72
  5057.1 1856.45  5072.1 1860.86  5085.7  1862.3  5114.2 1861.52  5135.2 1857.36
  5165.2 1854.58  5554.9  1856.7  5582.6 1857.43  5597.6  1859.9  5633.1 1859.29
#Mann= 5 ,-1 , 0
  4094.5     .07       0  4497.7    .033       0  4503.4     .07       0
  4506.1    .033       0  5023.2     .07       0
Bank Sta=4497.7,4503.4
XS Rating Curve= 0 ,0
Exp/Cntr=0.3,0.1

Type RM Length L Ch R = 1 ,10642   ,537,537,537
BEGIN DESCRIPTION:
Elm 01 31 10642.03
END DESCRIPTION:
XS GIS Cut Line= 3
      1550626.25      6819316.55      1550963.02      6818934.64
      1551459.56      6818108.23
#Sta/Elev= 30
  4499.4 1857.24  4766.4 1854.22  4780.7  1855.3  4816.7 1867.32  4837.6 1868.23
  4858.5 1865.04    4866 1861.01  4880.3 1856.42  4886.9 1857.62  4894.5 1854.96
  4908.7 1853.33  4969.4 1852.09  4969.9 1851.59  4975.1 1852.09    5028 1854.19
  5059.1 1858.17    5096 1860.32  5226.4 1859.37  5314.5 1858.79  5488.5 1859.14
    5504  1860.3  5509.8  1859.3  5525.4 1860.89  5540.9 1860.65  5546.8 1858.07
  5583.7 1859.65  5605.1 1858.56  5620.6 1855.45  5657.5 1854.05  5972.7 1856.35
#Mann= 5 ,-1 , 0
  4499.4     .07       0  4969.4     .07       0  4975.1     .07       0
  5226.4    .033       0  5314.5     .07       0
Bank Sta=4969.4,4975.1
XS Rating Curve= 0 ,0
Exp/Cntr=0.3,0.1

Type RM Length L Ch R = 1 ,10105   ,54,54,54
BEGIN DESCRIPTION:
Elm 01 31 10105.04
END DESCRIPTION:
XS GIS Cut Line= 4
      1550945.66       6819302.7      1551324.13      6819118.67
      1551456.08      6819045.75      1551719.96      6818205.51
#Sta/Elev= 30
  4423.7 1853.76  4645.4 1848.93  4689.8 1846.31    4702 1847.75  4741.5 1848.66
  4747.1 1850.69  4764.1 1849.61  4769.6 1852.81  4786.6 1850.87  4792.2  1853.8
  4853.8 1848.38  4875.5 1847.71    4903  1842.4  4913.3 1843.37    4919 1846.72
  4940.8 1844.59  4962.6 1846.21  4978.6 1843.69  5021.5 1842.29    5022 1841.79
  5027.3 1842.29  5073.3 1842.62  5078.6 1843.73  5245.9 1849.94  5265.5 1849.24
  5317.9 1851.36  5337.9 1850.93  5343.1 1852.09  5391.2 1853.66    5876 1858.41
#Mann= 3 ,-1 , 0
  4423.7     .07       0  5021.5     .07       0  5027.3     .07       0
Bank Sta=5021.5,5027.3
XS Rating Curve= 0 ,0
Exp/Cntr=0.3,0.1

Type RM Length L Ch R = 1 ,10051   ,400,400,400
BEGIN DESCRIPTION:
Elm 01 31 10050.72
END DESCRIPTION:
XS GIS Cut Line= 3
      1550973.43       6819490.2       1551490.8      6819087.42
      1551806.78      6818583.93
#Sta/Elev= 30
  4335.9 1854.01  4553.1 1849.21  4609.2 1848.99  4638.2 1848.01  4837.2 1845.33
  4872.5 1846.16  4895.1 1845.79  4915.9 1844.84  4936.8 1842.06  4944.9 1842.28
  4951.2 1844.59  4958.9 1844.95    4972 1844.18  4991.1 1841.59  4999.8 1841.56
  5000.3 1841.06  5005.6 1841.56    5024 1842.94    5030 1844.49  5051.2 1845.86
  5087.7 1844.58  5118.3 1844.85  5145.4 1847.47  5203.4 1849.93  5349.2 1850.81
  5379.9 1851.67  5385.8 1851.12  5451.3 1854.36  5486.7 1855.33    5586  1853.5
#Mann= 3 ,-1 , 0
  4335.9     .07       0  4999.8     .07       0  5005.6     .07       0
Bank Sta=4999.8,5005.6
XS Rating Curve= 0 ,0
Exp/Cntr=0.3,0.1

Type RM Length L Ch R = 1 ,9651    ,317,317,317
BEGIN DESCRIPTION:
Elm 01 31 9650.51
END DESCRIPTION:
XS GIS Cut Line= 3
      1551046.37      6819535.33      1551601.91      6819448.53
      1552750.64      6819184.77
#Sta/Elev= 30
  4424.3 1852.27  4632.1 1848.16  4767.7  1846.9  4908.7 1842.59  4939.1 1841.95
  4979.6 1842.15  4990.7 1841.65    5000 1840.06  5013.3 1840.32  5017.5 1839.73
    5018 1839.23  5023.1 1839.23  5023.6 1839.73  5051.1 1841.64  5082.1 1841.97
  5246.3 1840.78  5256.5 1841.83  5275.6 1841.88  5318.1 1843.53  5441.2 1846.67
  5492.5 1849.06  5584.8 1849.45  5639.1 1850.79  5724.8  1848.1  5759.3 1847.86
  5815.7 1848.49  5858.5 1848.14  5997.4 1849.91  6138.9 1849.93  6165.2 1850.55
#Mann= 3 ,-1 , 0
  4424.3     .07       0  5017.5     .07       0  5023.6     .07       0
Bank Sta=5017.5,5023.6
XS Rating Curve= 0 ,0
Exp/Cntr=0.3,0.1

Type RM Length L Ch R = 1 ,9334    ,186,186,186
BEGIN DESCRIPTION:
Elm 01 31 9334.1
END DESCRIPTION:
XS GIS Cut Line= 3
      1551150.53       6819663.8      1551737.33      6819712.42
        1552529.      6819698.53
#Sta/Elev= 30
  4394.9 1851.37  4539.9 1849.22    4570 1850.93  4600.1 1844.94  4626.3 1844.57
  4631.3 1842.78  4650.2 1844.16  4670.3 1849.47  4700.4 1851.27  4730.5 1846.76
  4740.6 1847.37  4760.6 1846.51  4790.7 1842.13  4850.9 1838.86  4887.7 1838.24
  4888.2 1837.74  4894.5 1838.24  4941.2 1839.87  4983.7 1839.58  4991.4 1838.35
  5001.4 1840.18  5031.4 1839.13  5091.4 1839.31  5141.4 1841.73  5181.4 1842.29
  5271.4 1841.99  5491.5 1844.18  5523.5 1845.73  5661.5 1847.83  5775.5    1848
#Mann= 3 ,-1 , 0
  4394.9     .07       0  4887.7     .07       0  4894.5     .07       0
Bank Sta=4887.7,4894.5
XS Rating Curve= 0 ,0
Exp/Cntr=0.3,0.1

Type RM Length L Ch R = 1 ,9148    ,196,196,196
BEGIN DESCRIPTION:
Elm 01 31 9178.38
END DESCRIPTION:
XS GIS Cut Line= 3
      1551099.78      6819712.28      1551783.76      6819878.94
      1552610.08      6820017.81
#Sta/Elev= 30
  4274.7 1852.92  4475.6 1851.04    4490 1849.55  4496.2 1846.44  4526.6 1841.55
  4531.7 1843.04    4558 1840.22  4573.4 1840.75  4578.6 1843.75  4588.9  1846.1
    4630 1849.37  4640.3 1849.26    4662 1843.27  4671.2 1842.28  4722.7 1843.51
  4740.2 1842.74  4753.5 1840.42    4782 1839.78  4948.8 1839.43  4969.7 1838.62
  4973.4 1836.45  4973.9 1835.95  4980.2 1836.45  4990.1 1838.67  5010.4  1839.6
  5091.5 1839.13  5125.4 1840.59  5306.7 1841.83  5548.2 1844.16  5816.6 1846.87
#Mann= 5 ,-1 , 0
  4274.7    .035       0  4973.4    .035       0  4980.2    .035       0
  5306.7     .07       0  5548.2    .035       0
Bank Sta=4973.4,4980.2
XS Rating Curve= 0 ,0
Exp/Cntr=0.3,0.1

Type RM Length L Ch R = 1 ,8952    ,283,283,283
BEGIN DESCRIPTION:
Elm 01 31 8866.75
END DESCRIPTION:
XS GIS Cut Line= 3
      1551282.56      6819888.62      1551935.38      6820027.52
       1552619.4       6820180.3
#Sta/Elev= 30
  4361.1 1852.07  4373.8 1852.52  4467.3  1849.6  4516.9 1848.94  4524.2 1847.51
  4529.3 1848.53  4537.4 1846.04  4568.1 1842.85  4588.5 1844.82  4629.4 1841.39
  4690.8 1840.18  4803.2 1838.52  4844.1 1838.72    4861 1839.75  4910.6 1838.51
    4977 1838.72  4997.5  1837.6  5004.7  1834.7  5009.8 1835.73  5014.5 1834.18
    5015 1833.68  5021.4 1834.18  5025.8 1837.86  5053.7 1839.16  5145.7  1838.6
  5181.8 1840.72  5237.7 1840.41    5356 1842.76  5632.7  1845.6  5729.4 1845.73
#Mann= 4 ,-1 , 0
  4361.1    .035       0  4467.3     .07       0  5014.5     .07       0
  5021.4     .07       0
Bank Sta=5014.5,5021.4
XS Rating Curve= 0 ,0
Exp/Cntr=0.3,0.1

Type RM Length L Ch R = 1 ,8669    ,210,210,210
BEGIN DESCRIPTION:
Elm 01 31 8669.19
END DESCRIPTION:
XS GIS Cut Line= 3
      1551258.12      6820059.62      1551963.02      6820292.28
       1552636.6      6820368.66
#Sta/Elev= 30
    4265 1852.71  4271.4 1851.75  4332.5 1850.08  4419.7 1848.05  4498.9  1845.1
  4662.9 1841.83  4689.4 1840.69  4872.5 1837.69  4935.7 1838.73  4967.3 1836.06
  4998.9 1836.39  5002.3 1833.23  5002.8 1832.73  5009.2 1833.23  5019.4 1834.35
  5029.4 1836.49  5039.5 1837.26  5059.6 1837.11  5089.8 1838.45  5140.1 1838.63
  5180.4 1840.05  5351.5 1841.44  5411.9 1842.64    5547 1842.89    5583 1844.02
  5603.1 1843.95  5613.1  1842.8  5663.5 1842.86  5673.5 1844.05  5685.2 1844.26
#Mann= 4 ,-1 , 0
    4265    .035       0  4332.5     .07       0  5002.3     .07       0
  5009.2     .07       0
Bank Sta=5002.3,5009.2
XS Rating Curve= 0 ,0
Exp/Cntr=0.3,0.1

Type RM Length L Ch R = 1 ,8459    ,362,362,362
BEGIN DESCRIPTION:
Elm 01 31 8459.37
END DESCRIPTION:
XS GIS Cut Line= 3
      1551278.98      6820208.94      1551824.13      6820358.25
      1552560.09      6820927.57
#Sta/Elev= 30
    4249  1850.6  4262.4 1849.91  4365.5 1847.77  4441.9 1845.69    4490 1843.59
  4628.5 1840.32  4701.1 1839.77  4857.1 1837.45  4871.6 1837.66  4878.5 1838.34
  4935.9 1836.36  4950.4  1836.8  4964.9 1836.13  4979.4 1836.22  4992.3 1836.73
  4996.8 1831.78  4997.3 1831.28  5003.2 1831.28  5003.7 1831.78    5021 1833.76
  5029.2  1837.1    5079 1836.17  5099.8 1836.91  5234.7 1839.12  5377.8 1839.67
  5384.3 1840.17  5413.1 1840.45  5556.2 1840.47  5727.4 1841.92  5744.7 1842.15
#Mann= 5 ,-1 , 0
    4249    .035       0  4365.5     .07       0  4996.8     .07       0
  5003.7     .07       0  5727.4    .035       0
Bank Sta=4996.8,5003.7
XS Rating Curve= 0 ,0
Exp/Cntr=0.3,0.1

Type RM Length L Ch R = 1 ,8097    ,239,239,239
BEGIN DESCRIPTION:
Elm 01 31 8097.46
END DESCRIPTION:
XS GIS Cut Line= 3
      1551390.12      6820372.15       1551803.3      6820747.14
      1552424.45      6821243.36
#Sta/Elev= 30
  4449.6 1847.17  4669.8 1840.57  4768.4 1838.44  4952.9 1837.25  4973.9  1835.5
  4998.8  1831.4  4999.3  1830.9  5005.2  1830.9  5005.7  1831.4  5007.6 1832.45
  5011.9 1832.45  5016.6  1834.3    5023 1834.42  5080.6  1834.1    5087 1832.99
    5095  1832.9  5115.8 1833.62  5123.8 1833.09  5130.2 1833.76  5137.7 1832.97
  5144.6 1833.73    5151 1833.39  5179.9 1834.66  5237.5 1834.51  5251.9 1833.71
  5279.1  1837.2  5329.7 1836.99  5386.4 1838.05  5514.5 1837.86  5802.6 1840.24
#Mann= 3 ,-1 , 0
  4449.6     .05       0  4998.8     .07       0  5005.7     .05       0
#XS Ineff= 2 , 0
       0                    5180       0    1837
Permanent Ineff=
       F       F
Bank Sta=4998.8,5005.7
XS Rating Curve= 0 ,0
Exp/Cntr=0.3,0.1

Type RM Length L Ch R = 1 ,7858    ,313,313,313
BEGIN DESCRIPTION:
Elm 01 31 7817.94
END DESCRIPTION:
XS GIS Cut Line= 3
      1551223.63      6820564.77      1551692.35      6820929.32
      1552361.27      6821449.21
#Sta/Elev= 30
  4355.7 1850.13  4451.5 1848.54  4565.5 1844.75  4594.5 1842.97  4600.8 1843.76
    4609  1842.3  4615.3 1842.88  4644.2 1840.75  4700.4 1838.93  4800.8 1836.56
  4907.6 1835.81  4914.9 1829.99  4924.8 1828.19  4925.3 1827.69  4931.9 1828.19
  4936.5 1829.36  4942.9 1829.43    4948 1833.23  4952.5 1833.23  4957.3 1831.71
  4965.5 1833.87  4971.8    1832  4978.2 1835.38  5000.8 1833.91  5036.1 1835.14
  5079.5 1834.24  5313.9 1836.61  5548.3  1837.5    5770  1840.3  5796.7 1841.61
#Mann= 3 ,-1 , 0
  4355.7    .035       0  4924.8    .035       0  4931.9    .035       0
Bank Sta=4924.8,4931.9
XS Rating Curve= 0 ,0
Exp/Cntr=0.3,0.1

Type RM Length L Ch R = 1 ,7545    ,419,419,419
BEGIN DESCRIPTION:
Elm 01 31 7544.79
END DESCRIPTION:
XS GIS Cut Line= 3
      1551070.67      6820813.11      1551584.55        6821202.
      1552410.48      6821649.67
#Sta/Elev= 30
  4351.8 1850.65  4420.4  1849.6    4601 1844.58  4771.6  1834.5  4808.7 1834.22
  4836.1 1831.76  4844.4 1832.27  4850.7 1830.86  4865.2 1833.73  4871.5 1832.82
  4886.1 1833.99  4894.3 1833.19  4900.6 1834.51  4908.9 1833.31  4958.8 1833.53
  4971.7 1832.56  4979.7 1830.34  5000.4 1831.16  5004.6  1830.3  5005.1  1829.8
  5011.7  1830.3  5022.3 1830.31  5060.3  1834.7  5142.1 1833.19  5531.4 1836.67
    5628 1836.34  5795.1  1839.3  5908.5 1841.01  5914.2 1841.24  5935.7 1841.71
#Mann= 7 ,-1 , 0
  4351.8    .035       0  4420.4     .07       0  5004.6     .07       0
  5011.7     .07       0  5795.1    .035       0  5908.5    .063       0
  5914.2    .035       0
Bank Sta=5004.6,5011.7
XS Rating Curve= 0 ,0
Exp/Cntr=0.3,0.1

Type RM Length L Ch R = 1 ,7126    ,116,116,116
BEGIN DESCRIPTION:
Elm 01 31 7126.25
END DESCRIPTION:
XS GIS Cut Line= 3
      1550931.75      6821351.29      1551501.22      6821573.53
      1552279.02      6821712.42
#Sta/Elev= 30
  4385.9 1839.42  4400.1 1840.36  4449.1 1837.44  4639.9 1832.55  4718.7 1832.14
  4773.1 1830.71  4832.8 1831.73  4881.8 1829.62    4917 1829.09  4926.1  1829.9
  5011.2 1829.71  5031.5 1827.83  5048.9 1830.82  5072.1 1831.26  5092.5 1833.99
  5102.6 1834.18  5133.1 1827.83  5153.4 1825.22  5170.1 1824.72  5170.6 1824.22
  5177.3 1824.72  5204.2 1830.67  5214.4 1832.16  5397.3 1833.45  5417.5 1834.74
  5437.8 1834.07  5498.8 1835.31  5558.9 1835.33  5722.3  1837.9  5787.3 1839.74
#Mann= 4 ,-1 , 0
  4385.9    .035       0  4449.1     .07       0  5170.1     .07       0
  5177.3     .07       0
Bank Sta=5170.1,5177.3
XS Rating Curve= 0 ,0
Exp/Cntr=0.3,0.1

Type RM Length L Ch R = 1 ,7010    ,288,288,288
BEGIN DESCRIPTION:
Elm 01 31 7010.02
END DESCRIPTION:
XS GIS Cut Line= 3
      1550924.87      6821483.26      1551424.83      6821660.33
      1552131.58      6821837.02
#Sta/Elev= 30
  4463.8 1837.86  4500.2 1836.86  4584.4 1835.09  4640.9 1832.79  4728.2 1831.37
  4882.7 1830.81  4898.9 1828.11  4916.5 1826.62    4917 1826.12  4923.7 1826.62
  4930.7 1827.84  4962.5 1828.27  4975.3 1827.28  5007.5 1827.73  5043.6 1830.11
  5066.5 1829.59  5097.4 1834.11  5126.1  1834.8  5179.9 1834.13  5208.5 1835.68
  5213.7 1834.23  5249.7 1835.95  5254.9 1834.42    5283 1835.77  5344.8 1836.21
  5355.1 1836.08  5365.4 1833.89  5386.1 1832.64  5602.5 1834.85  5722.7 1837.53
#Mann= 4 ,-1 , 0
  4463.8    .035       0  4500.2     .07       0  4916.5     .07       0
  4923.7     .07       0
Bank Sta=4916.5,4923.7
XS Rating Curve= 0 ,0
Exp/Cntr=0.3,0.1

Type RM Length L Ch R = 1 ,6722    ,111,111,111
BEGIN DESCRIPTION:
Elm 01 31 6721.62
END DESCRIPTION:
XS GIS Cut Line= 3
      1550886.65      6821767.97      1551414.41      6821917.28
       1552004.7       6822052.7
#Sta/Elev= 30
  4460.4 1834.88  4577.2 1833.33  4926.3 1830.22  4965.4  1828.4  4978.3 1827.23
  4995.4 1823.91  4995.9 1823.41  5002.7 1823.91  5019.7  1824.9  5029.7 1828.86
  5083.7 1827.81  5091.6 1827.88  5120.6 1834.66  5125.7 1831.65  5142.9 1832.43
  5163.4 1829.19  5168.6 1831.79  5173.7 1829.83  5211.5 1833.27  5216.6 1828.97
  5235.2 1829.81  5254.3 1832.62  5259.5 1829.96  5276.2 1831.76  5286.5 1829.67
  5296.8 1829.13  5339.5  1830.1  5501.9 1832.59  5569.9 1835.49  5614.5 1835.72
#Mann= 7 ,-1 , 0
  4460.4    .035       0  4577.2     .07       0  4965.4    .035       0
  4995.4    .035       0  5002.7    .035       0  5083.7     .07       0
  5339.5    .035       0
Bank Sta=4995.4,5002.7
XS Rating Curve= 0 ,0
Exp/Cntr=0.3,0.1

Type RM Length L Ch R = 1 ,6611    ,279,279,279
BEGIN DESCRIPTION:
Elm 01 31 6528.6
END DESCRIPTION:
XS GIS Cut Line= 3
       1550772.8      6821941.06      1551387.34      6822020.92
      1552031.62      6822187.18
#Sta/Elev= 30
  4363.6 1835.42  4458.9 1833.47  4527.2 1833.57  4547.3 1832.31  4612.2 1831.43
  4683.5 1831.41    4815 1829.72  4923.7 1829.43  4940.6 1828.55    4976 1823.35
  4976.5 1822.85  4983.3 1823.35    4994 1823.64  5011.9 1825.96  5034.7  1824.2
  5053.2 1826.29  5094.5 1826.09    5117 1827.32  5192.2 1826.76  5249.4 1827.92
  5268.3 1829.37  5273.5 1828.75  5404.3 1832.05    5431 1831.59  5471.7 1832.65
  5476.8 1833.56  5507.2 1832.85  5579.9 1835.45  5593.7 1834.85  5648.7    1836
#Mann= 6 ,-1 , 0
  4363.6     .07       0  4683.5    .035       0    4815     .07       0
    4976     .07       0  4983.3     .07       0    5117    .035       0
Bank Sta=4976,4983.3
XS Rating Curve= 0 ,0
Exp/Cntr=0.3,0.1

Type RM Length L Ch R = 1 ,6332    ,253,253,253
BEGIN DESCRIPTION:
Elm 01 31 6331.59
END DESCRIPTION:
XS GIS Cut Line= 3
      1550733.84      6822104.77      1551310.25      6822274.92
      1551966.54      6822524.93
#Sta/Elev= 30
  4403.1 1833.51  4431.3  1833.8  4497.9 1831.41  4541.6  1831.9  4613.4 1829.64
  4685.8 1830.06  4713.3 1829.03  4956.9 1826.85  5000.3 1821.98  5000.8 1821.48
  5007.7 1821.98  5031.4  1823.6  5050.8 1826.63  5073.4 1826.38  5080.9 1828.02
  5086.2  1825.4    5111 1828.61  5116.3 1827.94    5159 1828.55  5165.8  1826.4
  5180.4 1828.36  5201.8 1826.92  5250.7 1826.05  5275.5 1827.11  5319.5 1826.84
  5351.6 1828.81  5522.8 1831.35  5629.8 1834.27  5675.4 1833.88  5706.4  1834.6
#Mann= 3 ,-1 , 0
  4403.1     .07       0  5000.3     .07       0  5007.7     .07       0
Bank Sta=5000.3,5007.7
XS Rating Curve= 0 ,0
Exp/Cntr=0.3,0.1

Type RM Length L Ch R = 1 ,6079    ,42,42,42
BEGIN DESCRIPTION:
Elm 01 31 6078.62
END DESCRIPTION:
XS GIS Cut Line= 3
      1550674.85      6822229.79      1551185.25      6822465.89
      1551994.25      6822670.74
#Sta/Elev= 30
  4443.4 1831.92  4764.6 1827.52  4907.7 1828.71  4993.9 1826.84  4999.4 1824.44
  5002.9 1825.95  5026.1 1826.03    5033 1821.84  5046.8 1818.57    5074 1816.84
  5098.3 1818.96  5120.2 1817.38  5139.6 1813.31  5208.1 1811.86  5208.6 1811.36
  5215.5 1811.86  5217.2  1812.1    5238 1814.02  5428.4  1812.4    5443  1813.5
  5449.1 1817.22  5457.2 1819.31  5490.3  1828.9  5519.9 1833.13  5531.6 1830.59
  5552.2 1829.83  5696.7 1833.66  5775.1 1833.69  5823.4 1834.42  5840.3 1834.37
#Mann= 7 ,-1 , 0
  4443.4     .07       0  5208.1     .07       0  5215.5     .07       0
  5217.2     .16       0  5457.2     .07       0  5775.1    .035       0
  5823.4     .07       0
Bank Sta=5208.1,5215.5
XS Rating Curve= 0 ,0
Exp/Cntr=0.3,0.1

Type RM Length L Ch R = 1 ,6037    ,120,120,120
BEGIN DESCRIPTION:
Elm 01 31 5.0
END DESCRIPTION:
XS GIS Cut Line= 4
      1550709.31      6822290.39       1551219.7      6822526.49
      1551334.29      6822555.51      1551938.98      6822905.43
#Sta/Elev= 30
  4507.5 1831.26  4779.7 1827.09  4899.9 1826.99  4917.3 1829.56  4994.9 1824.79
  4995.4 1824.29  5002.3 1824.79  5042.9 1829.07  5060.4 1827.12  5065.7 1829.25
  5097.5 1828.61  5134.6 1826.16  5147.5 1830.35  5175.6 1827.06  5180.7 1831.55
  5198.8 1828.41  5204.6 1832.83  5220.4 1829.07  5226.2 1833.17  5241.9  1829.3
  5247.7 1833.43  5257.7 1831.63  5263.5 1834.28    5485 1831.84  5547.6 1828.64
  5616.4 1829.79    5638  1827.2  5681.1 1832.92  5686.8 1830.98  5886.7 1831.63
#Mann= 5 ,-1 , 0
  4507.5     .07       0  4994.9     .07       0  5002.3     .07       0
  5097.5     .16       0    5485     .07       0
Bank Sta=4994.9,5002.3
XS Rating Curve= 0 ,0
Exp/Cntr=0.3,0.1

Type RM Length L Ch R = 1 ,5917    ,201,201,201
BEGIN DESCRIPTION:
Elm 01 31 4.5
END DESCRIPTION:
XS GIS Cut Line= 4
      1550634.94      6822349.33      1551145.34      6822585.44
      1551259.94      6822614.45      1551863.49      6822963.72
#Sta/Elev= 30
  4376.8 1830.86  4859.4 1825.89  4927.8 1825.52  4933.3 1819.85  4936.3 1825.35
  4941.6 1825.35  4959.4 1820.54  4967.3 1823.87  4972.4 1820.98  4980.1 1823.99
  5086.3  1824.5  5144.1 1819.75  5189.4 1825.94  5210.9 1822.22  5216.7 1823.45
  5232.5 1817.33  5238.2 1818.63    5254 1814.91  5266.1 1814.53  5266.6 1814.03
  5273.5 1814.53  5291.3 1816.05  5297.1 1819.08  5334.4 1828.44  5386.7 1826.04
  5430.5 1828.62  5436.3 1827.07  5469.8 1827.86  5726.8 1831.18  5754.7 1830.99
#Mann= 6 ,-1 , 0
  4376.8     .07       0  4859.4     .16       0  5266.1     .07       0
  5273.5     .16       0  5469.8     .07       0  5726.8    .035       0
Bank Sta=5266.1,5273.5
XS Rating Curve= 0 ,0
Exp/Cntr=0.3,0.1

Type RM Length L Ch R = 1 ,5716    ,251,251,251
BEGIN DESCRIPTION:
Elm 01 31 5716.07
END DESCRIPTION:
XS GIS Cut Line= 3
      1550494.27      6822597.83      1551105.38       6822764.5
      1551848.43      6823035.33
#Sta/Elev= 30
  4366.7 1828.18  4771.7 1824.56    4801  1825.8  4813.2 1824.57  4927.2 1822.92
  4937.5 1820.94  4947.9 1821.07  4954.8 1822.95  4965.1  1822.2  4997.3 1819.79
  5042.3 1821.57  5117.3 1820.83  5127.5 1821.31  5148.7 1825.52  5167.8 1825.66
  5180.7 1823.88  5198.4 1819.15  5203.7  1821.4  5219.8 1821.06  5234.3 1820.74
  5265.8    1814    5294  1812.1  5294.5  1811.6  5301.4  1812.1  5315.3 1812.36
  5340.3 1815.44  5361.6 1821.13  5468.2  1826.8  5712.8 1830.49    5791 1829.92
#Mann= 5 ,-1 , 0
  4366.7     .07       0  4965.1     .16       0  5219.8     .07       0
    5294     .07       0  5301.4     .07       0
Bank Sta=5294,5301.4
XS Rating Curve= 0 ,0
Exp/Cntr=0.3,0.1

Type RM Length L Ch R = 1 ,5465    ,345,345,345
BEGIN DESCRIPTION:
Elm 01 31 5465.11
END DESCRIPTION:
XS GIS Cut Line= 3
      1550331.11      6822663.82      1551046.36      6822993.67
      1551827.65       6823278.4
#Sta/Elev= 30
  4210.2 1827.96  4335.6 1826.32  4390.7 1826.77  4523.5 1824.39  4621.9 1824.62
  4689.7 1822.76  4743.1 1823.23  4758.5 1821.69    4776 1823.33  4787.1 1823.37
  4832.9 1819.92  4930.3 1818.85  4993.5 1820.14    4997 1818.08  5003.3 1817.39
  5003.8 1816.89  5010.8 1817.39  5017.7 1819.54  5049.3 1818.65  5070.9 1819.02
  5134.8 1821.85    5156 1823.63  5288.5 1823.65  5349.6 1824.65  5374.9 1825.85
    5436 1825.17  5491.8 1827.28  5539.2 1826.41  5669.9 1828.41  5829.4 1828.83
#Mann= 3 ,-1 , 0
  4210.2     .07       0  5003.3     .07       0  5010.8     .07       0
Bank Sta=5003.3,5010.8
XS Rating Curve= 0 ,0
Exp/Cntr=0.3,0.1
