--- Elm 01 74.prj (project) ---

Proj Title=Elm 01 74 Base Level Engineering
Current Plan=p01
Default Exp/Contr=0.3,0.1
English Units
Geom File=g01
Flow File=f01
Plan File=p01
BEGIN DESCRIPTION:
Elm 01 74
END DESCRIPTION:

--- Elm 01 74.p01 (plan) ---

Plan Title=Multiple Run
Short Identifier=Multiple
Geom File=g01
Flow File=f01
Subcritical Flow
K Sum by GR= 0
Std Step Tol= 0.01
Critical Tol= 0.01
Num of Std Step Trials= 20
Max Error Tol= 0.3
Flow Tol Ratio= 0.001
Split Flow NTrial= 30
Split Flow Tol= 0.02
Split Flow Ratio= 0.02
Log Output Level= 0
Friction Slope Method= 1
Unsteady Friction Slope Method= 2
Unsteady Bridges Friction Slope Method= 1
Parabolic Critical Depth
Global Vel Dist=  1 , 1 , 1
Global Log Level= 0
CheckData=True
Encroach Param= -1, 0, 0, 0
BEGIN DESCRIPTION:
Multiple Run
END DESCRIPTION:

--- Elm 01 74.f01 (steady flow) ---

Flow Title=Multiple
Number of Profiles=7
Profile Names=10-year,25-year,50-year,1pct_min,100-year,1pct_plu,500-year
River Rch & RM= Elm 01 74,Reach-1,19926
     346     500     633     498     798    1100    1290
River Rch & RM= Elm 01 74,Reach-1,18009
     477     694     884     697    1120    1540    1810
River Rch & RM= Elm 01 74,Reach-1,8170
     525     766     975     769    1230    1700    1990
Boundary for River Rch & Prof#=Elm 01 74,Reach-1,1
Up Type=0
Dn Type=3
Dn Slope=0.001
Boundary for River Rch & Prof#=Elm 01 74,Reach-1,2
Up Type=0
Dn Type=3
Dn Slope=0.001
Boundary for River Rch & Prof#=Elm 01 74,Reach-1,3
Up Type=0
Dn Type=3
Dn Slope=0.001
Boundary for River Rch & Prof#=Elm 01 74,Reach-1,4
Up Type=0
Dn Type=3
Dn Slope=0.001
Boundary for River Rch & Prof#=Elm 01 74,Reach-1,5
Up Type=0
Dn Type=3
Dn Slope=0.001
Boundary for River Rch & Prof#=Elm 01 74,Reach-1,6
Up Type=0
Dn Type=3
Dn Slope=0.001
Boundary for River Rch & Prof#=Elm 01 74,Reach-1,7
Up Type=0
Dn Type=3
Dn Slope=0.001

--- Elm 01 74.g01 (geometry) ---

Geom Title=Existing Conditions

River Reach=Elm 01 74,Reach-1
Reach XY= 30
      1588655.00      6777238.00      1588357.23      6776832.07
      1588311.51      6776195.62      1587960.93      6776285.77
      1587560.61      6776082.41      1587362.01      6775797.03
      1586882.20      6775687.44      1586751.66      6775780.40
      1586275.05      6775587.80      1585753.54      6776134.46
      1585060.86      6776140.07      1584753.54      6776484.46
      1583652.69      6776793.82      1583399.16      6777285.95
      1582324.98      6777338.04      1581949.48      6777140.35
      1581556.46      6777141.54      1580944.57      6777936.95
      1580420.16      6777888.39      1579825.21      6778038.21
      1579344.56      6777789.05      1578510.94      6777785.74
      1577106.47      6777284.45      1576740.96      6776938.09
      1576525.15      6777038.37      1573879.78      6776987.67
      1573751.69      6777379.98      1573556.28      6777449.03
      1573497.52      6777894.06      1573055.00      6778238.00

Type RM Length L Ch R = 1,19926,292,292,292
BEGIN DESCRIPTION:
Elm 01 74 19642.71
END DESCRIPTION:
XS GIS Cut Line= 3
      1589203.47      6776853.74      1588642.41      6777225.60
      1588168.56      6777637.12
#Sta/Elev= 30
  4326.9 2139.41  4394.5 2133.43  4482.7 2128.55  4544.9 2125.09  4553.0 2122.12
  4653.2 2120.44  4776.8 2112.85  4804.2 2111.39  4926.9 2104.09  4942.0 2102.31
  4957.0 2095.45  4972.0 2092.07  4991.1 2090.84  4991.3 2090.34  4995.1 2090.84
  5028.1 2091.84  5056.6 2099.28  5220.0 2108.46  5261.7 2117.40  5269.3 2116.70
  5288.5 2118.71  5304.4 2119.22  5326.3 2117.42  5368.1 2120.25  5453.5 2121.49
  5468.2 2122.95  5531.4 2126.76  5574.1 2126.58  5595.0 2130.16  5627.6 2132.34
#Mann=8,-1,0
  4326.9    0.12       0  4482.7    0.05       0  4776.8    0.12       0
  4804.2    0.05       0  4991.1    0.05       0  4995.1    0.05       0
  5288.5    0.12       0  5468.2    0.05       0
Bank Sta=4991.1,4995.1
Exp/Cntr=0.3,0.1

Type RM Length L Ch R = 1,19634,77,77,77
BEGIN DESCRIPTION:
Elm 01 74 19634.42
END DESCRIPTION:
XS GIS Cut Line= 4
      1589135.81      6776725.23      1588467.39      6777001.28
      1588373.64      6777051.63      1588061.15      6777518.63
#Sta/Elev= 30
  4278.0 2135.61  4333.0 2129.18  4447.9 2120.78  4456.5 2121.31  4527.7 2116.52
  4563.0 2115.67  4664.0 2107.27  4823.8 2103.50  4863.1 2099.89  4906.4 2090.39
  4930.3 2088.50  5027.1 2085.82  5027.4 2085.32  5031.1 2085.82  5060.6 2087.00
  5089.2 2095.17  5104.0 2097.49  5147.7 2098.30  5183.8 2101.82  5189.8 2103.40
  5225.8 2103.84  5240.8 2106.96  5255.8 2105.93  5306.9 2108.02  5442.0 2115.96
  5500.3 2118.03  5508.0 2119.39  5572.5 2121.00  5622.1 2126.70  5669.5 2128.86
#Mann=4,-1,0
  4278.0    0.12       0  4447.9    0.05       0  5027.1    0.05       0
  5031.1    0.05       0
Bank Sta=5027.1,5031.1
Exp/Cntr=0.3,0.1

Type RM Length L Ch R = 1,19557,75,75,75
BEGIN DESCRIPTION:
Elm 01 74 19556.99
END DESCRIPTION:
XS GIS Cut Line= 4
      1589116.70      6776622.81      1588410.10      6776947.46
      1588253.85      6777023.85      1587809.34      6777442.41
#Sta/Elev= 30
  4227.3 2135.94  4317.2 2126.71  4369.1 2125.32  4375.8 2123.68  4466.5 2115.50
  4526.3 2114.21  4564.0 2109.50  4677.9 2103.38  4701.1 2102.25  4768.4 2100.03
  4810.4 2096.02  4810.7 2095.52  4814.4 2096.02  4834.4 2100.78  4856.5 2102.78
  5055.1 2103.22  5061.9 2101.92  5067.4 2103.37  5188.2 2104.37  5195.0 2102.66
  5230.6 2102.22  5280.0 2105.65  5294.2 2108.52  5421.6 2113.59  5428.5 2112.15
  5442.6 2115.24  5506.6 2116.19  5534.5 2118.51  5633.6 2120.99  5789.4 2128.28
#Mann=6,-1,0
  4227.3    0.12       0  4375.8    0.05       0  4677.9    0.12       0
  4701.1    0.05       0  4810.4    0.05       0  4814.4    0.05       0
Bank Sta=4810.4,4814.4
Exp/Cntr=0.3,0.1

Type RM Length L Ch R = 1,19482,195,195,195
BEGIN DESCRIPTION:
Elm 01 74 19482.41
END DESCRIPTION:
XS GIS Cut Line= 4
      1589073.27      6776532.54      1588387.53      6776878.01
      1588222.60      6776954.40      1587679.58      6777207.70
#Sta/Elev= 30
  4235.7 2133.21  4260.4 2131.17  4277.1 2128.07  4334.8 2124.43  4371.9 2126.18
  4424.1 2124.05  4446.5 2122.00  4468.9 2115.43  4513.7 2110.04  4577.7 2106.77
  4726.7 2097.89  4834.8 2091.92  4857.1 2091.23  4862.7 2092.61  4885.0 2088.56
  4901.8 2088.15  4907.4 2089.74  4924.1 2085.70  4989.0 2083.15  4989.2 2082.65
  4993.0 2083.15  5065.0 2087.33  5105.3 2088.01  5139.2 2091.92  5156.6 2096.53
  5215.8 2103.24  5487.8 2111.20  5516.2 2114.17  5556.4 2113.67  5784.5 2117.73
#Mann=6,-1,0
  4235.7    0.12       0  4334.8    0.05       0  4577.7    0.12       0
  4726.7    0.05       0  4989.0    0.05       0  4993.0    0.05       0
Bank Sta=4989,4993
Exp/Cntr=0.3,0.1

Type RM Length L Ch R = 1,19287,223,223,223
BEGIN DESCRIPTION:
Mapping XS 0756ffd4
END DESCRIPTION:
XS GIS Cut Line= 4
      1588915.88      6776488.33      1588510.02      6776661.96
      1588154.12      6776735.74      1587869.88      6776915.83
#Sta/Elev= 30
  4403.5 2119.19  4433.9 2116.93  4494.3 2113.01  4502.4 2110.61  4538.6 2108.82
  4632.9 2106.83  4693.9 2097.88  4709.0 2097.83  4800.0 2091.62  4852.6 2088.77
  4897.7 2079.82  4911.3 2083.41  4921.6 2083.14  4947.8 2079.07  5001.3 2078.07
  5001.5 2077.57  5005.3 2078.07  5023.7 2078.46  5033.9 2081.97  5043.1 2087.64
  5048.2 2087.72  5054.3 2093.33  5064.5 2097.94  5074.7 2099.36  5166.7 2102.25
  5238.8 2108.78  5275.3 2108.80  5332.9 2104.82  5499.8 2105.60  5544.9 2106.88
#Mann=6,-1,0
  4403.5    0.12       0  4433.9    0.05       0  4538.6    0.12       0
  4800.0    0.05       0  5001.3    0.05       0  5005.3    0.05       0
Bank Sta=5001.3,5005.3
Exp/Cntr=0.3,0.1

Type RM Length L Ch R = 1,19064,45,45,45
BEGIN DESCRIPTION:
Elm 01 74 19063.94
END DESCRIPTION:
XS GIS Cut Line= 3
      1588519.91      6776453.64      1588354.95      6776516.15
      1588229.53      6776575.84
#Sta/Elev= 30
  4824.5 2091.58  4861.8 2088.32  4893.9 2087.16  4903.3 2085.94  4915.3 2081.34
  4919.3 2081.03  4926.0 2080.52  4933.5 2078.84  4938.8 2073.74  4947.4 2072.18
  4956.1 2071.67  4956.3 2071.17  4960.1 2071.67  4963.6 2072.51  4969.0 2071.89
  4988.4 2075.19  4993.8 2074.28  4998.2 2077.03  5003.6 2077.03  5011.6 2081.90
  5017.1 2086.12  5023.0 2088.32  5039.9 2092.63  5062.6 2093.16  5068.1 2094.25
  5078.4 2094.08  5100.5 2097.99  5130.7 2097.81  5136.2 2098.49  5139.8 2097.70
#Mann=4,-1,0
  4824.5    0.12       0  4919.3    0.05       0  4956.1    0.05       0
  4960.1    0.05       0
Bank Sta=4956.1,4960.1
Exp/Cntr=0.3,0.1

Type RM Length L Ch R = 1,19019,47,47,47
BEGIN DESCRIPTION:
Elm 01 74 19018.74
END DESCRIPTION:
XS GIS Cut Line= 3
      1588478.19      6776411.13      1588338.46      6776475.35
      1588220.15      6776543.08
#Sta/Elev= 30
  4847.0 2088.24  4876.7 2086.67  4886.9 2085.57  4899.7 2085.23  4905.5 2084.46
  4936.6 2083.72  4936.8 2083.22  4940.3 2083.22  4940.6 2083.72  4960.6 2085.77
  4968.6 2087.48  4974.1 2084.70  4982.6 2087.19  4991.6 2088.15  4997.1 2086.27
  4999.9 2087.91  5005.7 2087.91  5013.4 2086.68  5019.1 2088.42  5027.8 2087.44
  5034.9 2085.62  5040.7 2089.69  5056.5 2090.14  5062.4 2093.09  5072.3 2096.27
  5078.1 2096.27  5085.4 2097.08  5108.5 2096.40  5131.3 2097.24  5137.1 2097.10
#Mann=4,-1,0
  4847.0    0.12       0  4886.9    0.05       0  4936.6    0.05       0
  4940.6    0.05       0
Bank Sta=4936.6,4940.6
Exp/Cntr=0.3,0.1

Type RM Length L Ch R = 1,18972,278,278,278
BEGIN DESCRIPTION:
Elm 01 74 18972.49
END DESCRIPTION:
XS GIS Cut Line= 3
      1588468.64      6776352.11      1588308.94      6776439.76
      1588178.97      6776528.42
#Sta/Elev= 30
  4819.7 2087.31  4835.3 2086.61  4841.7 2085.79  4863.4 2085.41  4879.5 2083.91
  4885.2 2084.25  4901.3 2082.67  4907.0 2083.35  4928.8 2082.71  4937.9 2081.84
  4944.9 2079.56  4950.6 2079.14  4964.7 2074.28  4965.0 2073.78  4968.5 2073.78
  4968.7 2074.28  4972.4 2075.04  4982.8 2074.43  4988.5 2076.44  4995.0 2075.14
  5001.3 2074.90  5018.7 2076.21  5025.1 2080.73  5031.1 2082.95  5040.0 2089.44
  5054.9 2094.82  5111.8 2094.88  5139.8 2096.00  5147.7 2095.29  5159.2 2095.67
#Mann=3,-1,0
  4819.7    0.05       0  4964.7    0.05       0  4968.7    0.05       0
Bank Sta=4964.7,4968.7
Exp/Cntr=0.3,0.1

Type RM Length L Ch R = 1,18694,269,269,269
BEGIN DESCRIPTION:
Elm 01 74 18694.38
END DESCRIPTION:
XS GIS Cut Line= 3
      1588447.71      6775909.39      1588308.83      6776197.57
      1588169.98      6776508.25
#Sta/Elev= 30
  4683.0 2106.18  4768.6 2104.59  4870.2 2100.38  4892.4 2097.93  4913.1 2098.56
  4925.6 2096.10  4936.8 2089.86  4947.9 2086.40  4959.3 2077.86  4970.1 2072.68
  4976.4 2067.51  4980.0 2067.07  4980.2 2066.57  4984.0 2067.07  4992.3 2067.99
  5001.6 2071.73  5005.9 2071.73  5019.3 2075.53  5036.2 2079.67  5045.4 2080.30
  5112.9 2080.62  5149.2 2082.51  5166.9 2085.47  5172.4 2084.46  5195.6 2087.91
  5218.8 2089.11  5255.3 2087.96  5265.2 2091.37  5288.2 2094.17  5343.2 2094.99
#Mann=6,-1,0
  4683.0    0.12       0  4768.6    0.05       0  4913.1    0.12       0
  4980.0    0.07       0  4984.0    0.12       0  5019.3    0.05       0
Bank Sta=4980,4984
Exp/Cntr=0.3,0.1

Type RM Length L Ch R = 1,18425,239,239,239
BEGIN DESCRIPTION:
Elm 01 74 18424.53
END DESCRIPTION:
XS GIS Cut Line= 3
      1588088.72      6776087.74      1588078.30      6776286.98
      1588066.58      6776458.87
#Sta/Elev= 30
  4800.0 2084.51  4820.3 2083.81  4890.4 2082.37  4930.4 2081.30  4940.4 2079.76
  4944.5 2078.92  4950.5 2077.70  4966.2 2075.03  4971.2 2073.45  4990.5 2069.48
  4997.5 2066.92  5002.5 2066.92  5010.6 2063.86  5018.6 2062.03  5018.8 2061.53
  5022.3 2061.53  5022.6 2062.03  5030.6 2064.44  5040.6 2069.37  5060.7 2080.65
  5070.7 2085.40  5080.7 2087.20  5090.7 2087.56  5100.8 2088.31  5118.7 2089.23
  5123.7 2088.43  5140.9 2087.95  5150.9 2086.67  5168.9 2084.97  5171.8 2084.97
#Mann=4,-1,0
  4800.0    0.12       0  4944.5    0.05       0  5018.6    0.05       0
  5022.6    0.05       0
Bank Sta=5018.6,5022.6
Exp/Cntr=0.3,0.1

Type RM Length L Ch R = 1,18186,177,177,177
BEGIN DESCRIPTION:
Elm 01 74 18186.22
END DESCRIPTION:
XS GIS Cut Line= 3
      1587936.39      6776065.60      1587855.65      6776233.60
      1587797.06      6776402.85
#Sta/Elev= 30
  4814.1 2081.99  4831.8 2081.04  4839.0 2080.33  4853.8 2080.12  4870.9 2079.26
  4882.0 2077.96  4916.1 2075.60  4938.8 2073.31  4967.0 2068.44  4972.5 2068.73
  4983.2 2067.59  4989.6 2063.60  4995.1 2063.09  4998.2 2060.49  4998.4 2059.99
  5001.9 2059.99  5002.2 2060.49  5019.4 2061.29  5036.9 2064.02  5045.3 2066.14
  5050.6 2065.69  5058.1 2068.07  5076.4 2074.87  5081.7 2075.69  5100.4 2079.84
  5107.6 2080.81  5112.9 2080.40  5138.7 2082.18  5169.9 2083.46  5179.6 2083.14
#Mann=5,-1,0
  4814.1    0.05       0  4831.8    0.12       0  4882.0    0.05       0
  4998.2    0.05       0  5002.2    0.05       0
Bank Sta=4998.2,5002.2
Exp/Cntr=0.3,0.1

Type RM Length L Ch R = 1,18009,164,164,164
BEGIN DESCRIPTION:
Elm 01 74 18009.3
END DESCRIPTION:
XS GIS Cut Line= 3
      1587803.48      6775973.34      1587707.12      6776145.23
      1587623.80      6776311.01
#Sta/Elev= 30
  4803.9 2085.98  4857.2 2079.51  4872.3 2079.35  4884.2 2078.24  4915.7 2076.15
  4937.4 2073.24  4953.4 2072.53  4969.3 2069.16  4975.0 2069.21  4996.7 2064.15
  4999.7 2061.90  5005.3 2061.90  5016.8 2058.14  5017.1 2057.64  5020.8 2058.14
  5026.4 2059.06  5041.2 2063.73  5048.8 2064.52  5057.9 2062.40  5063.5 2062.03
  5080.2 2064.35  5085.8 2064.04  5093.6 2067.16  5102.5 2069.36  5108.1 2069.91
  5130.5 2075.30  5138.4 2076.39  5152.8 2077.62  5175.1 2077.29  5186.5 2077.88
#Mann=5,-1,0
  4803.9    0.05       0  4857.2    0.12       0  4884.2    0.05       0
  5016.8    0.05       0  5020.8    0.05       0
Bank Sta=5016.8,5020.8
Exp/Cntr=0.3,0.1

Type RM Length L Ch R = 1,17845,249,249,249
BEGIN DESCRIPTION:
Elm 01 74 17845.08
END DESCRIPTION:
XS GIS Cut Line= 3
      1587677.63      6775915.16      1587559.55      6776082.73
      1587479.98      6776182.62
#Sta/Elev= 30
  4796.3 2077.96  4807.7 2077.51  4813.8 2076.54  4836.5 2075.60  4843.4 2074.87
  4893.9 2071.76  4914.9 2068.61  4929.6 2065.65  4935.8 2065.76  4944.4 2064.40
  4965.4 2062.46  4971.5 2060.78  4980.6 2058.97  4998.9 2056.07  4999.2 2055.57
  5002.7 2055.57  5002.9 2056.07  5015.5 2057.95  5029.9 2057.81  5036.3 2059.58
  5044.4 2058.84  5050.7 2067.42  5058.8 2067.61  5065.2 2072.31  5079.6 2073.37
  5086.0 2075.61  5100.4 2077.15  5114.8 2078.21  5122.8 2078.28  5129.0 2079.07
#Mann=4,-1,0
  4796.3    0.12       0  4980.6    0.05       0  4998.9    0.05       0
  5002.9    0.05       0
Bank Sta=4998.9,5002.9
Exp/Cntr=0.3,0.1

Type RM Length L Ch R = 1,17596,306,306,306
BEGIN DESCRIPTION:
Elm 01 74 17596.08
END DESCRIPTION:
XS GIS Cut Line= 3
      1587572.41      6775731.46      1587409.68      6775890.93
      1587314.23      6776011.34
#Sta/Elev= 30
  4774.5 2075.97  4798.6 2074.65  4840.9 2073.84  4862.2 2072.44  4869.2 2070.77
  4876.3 2072.11  4883.3 2068.94  4890.4 2068.93  4897.4 2064.65  4903.9 2063.80
  4911.6 2060.91  4954.0 2057.69  4961.2 2056.31  4968.2 2057.06  4973.3 2054.90
  4973.6 2054.40  4977.1 2054.40  4977.4 2054.90  4978.4 2054.93  5017.8 2059.83
  5024.2 2058.93  5032.3 2059.54  5046.7 2061.72  5053.1 2065.78  5075.2 2069.07
  5096.4 2070.64  5102.7 2071.94  5117.2 2073.11  5146.0 2075.09  5156.0 2075.02
#Mann=4,-1,0
  4774.5    0.12       0  4973.3    0.05       0  4977.4    0.12       0
  4978.4    0.05       0
Bank Sta=4973.3,4977.4
Exp/Cntr=0.3,0.1

Type RM Length L Ch R = 1,17290,184,184,184
BEGIN DESCRIPTION:
Elm 01 74 17289.82
END DESCRIPTION:
XS GIS Cut Line= 3
      1587190.50      6775575.14      1587194.84      6775790.02
      1587195.92      6775980.99
#Sta/Elev= 30
  4785.7 2070.65  4789.6 2070.65  4798.6 2069.53  4818.6 2068.67  4838.6 2067.10
  4852.1 2065.45  4858.6 2064.22  4868.6 2061.54  4898.6 2059.10  4908.6 2057.62
  4958.6 2054.84  4968.6 2054.63  4978.6 2053.70  4988.6 2050.55  4995.1 2049.68
  4995.3 2049.18  4998.9 2049.18  4999.2 2049.68  5000.6 2049.68  5008.6 2052.51
  5028.6 2062.53  5038.6 2064.45  5058.6 2064.37  5078.6 2064.87  5108.6 2067.73
  5118.6 2067.75  5128.6 2068.33  5168.6 2068.85  5178.8 2068.51  5191.6 2068.99
#Mann=5,-1,0
  4785.7    0.05       0  4852.1    0.12       0  4995.1    0.07       0
  4999.2    0.12       0  5178.8    0.05       0
Bank Sta=4995.1,4999.2
Exp/Cntr=0.3,0.1

Type RM Length L Ch R = 1,17106,331,331,331
BEGIN DESCRIPTION:
Elm 01 74 17106.34
END DESCRIPTION:
XS GIS Cut Line= 3
      1586991.93      6775561.05      1587011.46      6775785.68
      1587020.07      6775955.68
#Sta/Elev= 30
  4774.2 2064.01  4801.3 2064.54  4821.3 2063.57  4831.4 2064.19  4841.4 2063.96
  4861.5 2060.16  4866.9 2058.29  4872.0 2058.98  4881.6 2057.51  4901.6 2055.77
  4921.7 2055.09  4951.8 2053.59  4971.9 2052.83  4979.9 2052.83  4984.9 2053.32
  4992.0 2052.75  4998.3 2051.09  5003.3 2051.09  5010.0 2048.54  5010.2 2048.04
  5013.8 2048.04  5014.1 2048.54  5022.0 2048.60  5032.0 2053.99  5042.1 2058.68
  5052.1 2062.94  5062.1 2063.63  5124.3 2064.27  5142.2 2064.28  5169.9 2065.75
#Mann=4,-1,0
  4774.2    0.12       0  5010.0    0.07       0  5014.1    0.12       0
  5124.3    0.05       0
Bank Sta=5010,5014.1
Exp/Cntr=0.3,0.1

Type RM Length L Ch R = 1,16775,257,257,257
BEGIN DESCRIPTION:
Elm 01 74 16775.22
END DESCRIPTION:
XS GIS Cut Line= 3
      1586765.41      6775577.61      1586752.39      6775780.72
      1586717.67      6775971.67
#Sta/Elev= 30
  4796.9 2060.53  4817.3 2060.66  4847.4 2060.26  4882.0 2059.49  4897.5 2058.51
  4907.5 2058.65  4927.6 2058.09  4947.6 2055.34  4957.6 2052.93  4977.7 2050.45
  4987.7 2048.65  4996.6 2046.25  5018.4 2045.06  5026.0 2044.99  5026.3 2044.49
  5030.0 2044.49  5030.2 2044.99  5038.3 2047.37  5048.5 2049.48  5071.8 2052.48
  5079.0 2054.39  5099.3 2061.20  5125.7 2067.79  5150.1 2072.12  5160.3 2072.83
  5170.4 2073.18  5178.5 2072.89  5183.6 2073.19  5190.1 2071.96  5194.5 2071.96
#Mann=4,-1,0
  4796.9    0.12       0  5026.0    0.07       0  5030.2    0.12       0
  5125.7    0.05       0
Bank Sta=5026,5030.2
Exp/Cntr=0.3,0.1

Type RM Length L Ch R = 1,16518,339,339,339
BEGIN DESCRIPTION:
Elm 01 74 16518.26
END DESCRIPTION:
XS GIS Cut Line= 3
      1586591.44      6775449.40      1586551.52      6775632.51
      1586510.73      6775888.57
#Sta/Elev= 30
  4814.1 2059.94  4843.4 2058.91  4868.4 2057.51  4884.3 2057.29  4894.5 2056.40
  4904.8 2053.10  4912.3 2047.82  4917.5 2048.09  4935.5 2050.35  4945.7 2049.73
  4956.0 2044.91  4959.2 2041.16  4959.5 2040.66  4963.2 2040.66  4963.5 2041.16
  4976.4 2042.83  4996.6 2046.33  5001.5 2046.33  5006.6 2049.65  5011.7 2049.54
  5017.2 2052.99  5027.3 2055.22  5037.5 2055.87  5088.1 2056.49  5136.0 2058.48
  5159.0 2058.90  5198.1 2060.98  5203.2 2060.75  5229.8 2062.27  5260.8 2063.36
#Mann=3,-1,0
  4814.1    0.12       0  4959.2    0.07       0  4963.5    0.12       0
Bank Sta=4959.2,4963.5
Exp/Cntr=0.3,0.1

Type RM Length L Ch R = 1,16179,259,259,259
BEGIN DESCRIPTION:
Elm 01 74 16179.48
END DESCRIPTION:
XS GIS Cut Line= 3
      1586156.58      6775440.71      1586256.38      6775593.45
      1586418.71      6775888.60
#Sta/Elev= 30
  4819.1 2074.07  4823.6 2073.53  4829.6 2071.72  4838.7 2071.65  4844.7 2070.48
  4851.7 2070.67  4859.8 2069.96  4874.9 2067.70  4947.0 2052.10  4974.4 2044.11
  4999.1 2038.06  4999.4 2037.56  5003.2 2037.56  5003.4 2038.06  5032.5 2039.14
  5048.6 2045.52  5054.3 2045.04  5086.5 2050.46  5092.2 2052.31  5098.1 2052.96
  5143.7 2054.68  5233.3 2056.07  5255.1 2057.28  5260.8 2056.77  5276.9 2057.88
  5282.6 2057.61  5298.7 2058.48  5320.5 2058.66  5326.3 2059.39  5338.4 2059.33
#Mann=4,-1,0
  4819.1    0.05       0  4947.0    0.12       0  4999.1    0.07       0
  5003.4    0.12       0
Bank Sta=4999.1,5003.4
Exp/Cntr=0.3,0.1

Type RM Length L Ch R = 1,15920,319,319,319
BEGIN DESCRIPTION:
Elm 01 74 15920.27
END DESCRIPTION:
XS GIS Cut Line= 3
      1585860.19      6775673.31      1586099.79      6775789.63
      1586331.24      6775959.77
#Sta/Elev= 30
  4734.5 2063.43  4751.0 2063.79  4756.6 2061.37  4762.2 2062.51  4779.2 2060.44
  4784.7 2060.89  4801.7 2058.27  4817.7 2058.90  4824.3 2056.39  4868.0 2053.53
  4937.1 2051.25  4942.7 2049.50  4959.7 2039.28  4971.1 2035.24  4971.4 2034.74
  4975.5 2035.24  5032.1 2038.84  5060.2 2039.05  5074.8 2040.51  5089.5 2046.80
  5095.7 2046.09  5104.1 2049.10  5110.3 2046.72  5118.8 2047.58  5125.0 2046.82
  5139.6 2049.62  5145.8 2048.80  5154.3 2049.36  5181.3 2052.85  5288.1 2058.12
#Mann=4,-1,0
  4734.5    0.05       0  4868.0    0.12       0  4971.1    0.07       0
  4975.5    0.12       0
Bank Sta=4971.1,4975.5
Exp/Cntr=0.3,0.1

Type RM Length L Ch R = 1,15601,207,207,207
BEGIN DESCRIPTION:
Elm 01 74 15601.48
END DESCRIPTION:
XS GIS Cut Line= 3
      1585762.97      6775794.82      1585906.21      6775993.63
      1586079.82      6776136.85
#Sta/Elev= 30
  4755.4 2052.52  4808.6 2050.43  4816.8 2049.23  4822.9 2050.08  4831.5 2050.13
  4852.4 2046.89  4858.5 2044.56  4867.1 2043.43  4873.2 2040.53  4881.8 2038.74
  4902.7 2036.16  4944.4 2034.32  4967.7 2034.46  4988.6 2035.30  5008.1 2034.15
  5008.4 2033.65  5012.2 2033.65  5012.5 2034.15  5059.8 2036.16  5074.1 2038.08
  5080.6 2039.92  5088.4 2040.36  5094.9 2043.23  5109.3 2044.69  5115.7 2046.67
  5123.6 2045.27  5130.1 2046.30  5137.9 2045.77  5193.9 2052.91  5225.5 2055.37
#Mann=3,-1,0
  4755.4    0.12       0  5008.1    0.07       0  5012.5    0.12       0
Bank Sta=5008.1,5012.5
Exp/Cntr=0.3,0.1

Type RM Length L Ch R = 1,15394,514,514,514
BEGIN DESCRIPTION:
Elm 01 74 15393.68
END DESCRIPTION:
XS GIS Cut Line= 3
      1585592.21      6775852.70      1585754.56      6776134.86
      1585907.33      6776336.23
#Sta/Elev= 30
  4675.4 2047.72  4710.7 2045.88  4716.5 2046.65  4726.5 2046.17  4732.3 2047.05
  4748.1 2045.51  4791.2 2043.82  4812.8 2044.47  4843.0 2043.60  4855.9 2042.40
  4865.9 2037.37  4871.7 2039.06  4900.7 2035.23  4909.0 2034.74  4914.8 2035.64
  4930.6 2032.43  4950.0 2031.61  4950.3 2031.11  4954.4 2031.61  4995.3 2032.50
  5054.2 2032.26  5075.0 2038.30  5081.3 2042.02  5089.6 2042.85  5095.8 2045.96
  5110.4 2048.01  5160.3 2051.01  5204.0 2052.43  5210.2 2053.65  5253.7 2054.58
#Mann=3,-1,0
  4675.4    0.12       0  4950.0    0.07       0  4954.4    0.12       0
Bank Sta=4950,4954.4
Exp/Cntr=0.3,0.1

Type RM Length L Ch R = 1,14880,341,341,341
BEGIN DESCRIPTION:
Elm 01 74 14880.16
END DESCRIPTION:
XS GIS Cut Line= 3
      1584969.45      6775659.43      1585258.49      6776094.30
      1585756.86      6776383.17
#Sta/Elev= 30
  4480.2 2110.22  4482.8 2106.69  4497.9 2104.84  4503.9 2101.20  4518.9 2097.23
  4622.6 2075.72  4642.2 2070.13  4663.2 2069.64  4714.3 2062.23  4735.4 2061.29
  4781.0 2052.79  4837.6 2041.17  4843.6 2045.63  4858.6 2043.68  4864.6 2047.12
  4930.8 2032.33  4936.8 2035.01  4981.9 2027.80  5065.4 2026.51  5065.7 2026.01
  5069.9 2026.51  5252.6 2029.77  5274.4 2034.87  5280.2 2038.81  5296.0 2035.65
  5360.6 2042.38  5435.1 2043.64  5440.9 2045.45  5449.1 2044.26  5578.4 2050.74
#Mann=5,-1,0
  4480.2    0.12       0  4622.6    0.05       0  4781.0    0.12       0
  5065.4    0.07       0  5069.9    0.12       0
Bank Sta=5065.4,5069.9
Exp/Cntr=0.3,0.1

Type RM Length L Ch R = 1,14539,338,338,338
BEGIN DESCRIPTION:
Elm 01 74 14539.03
END DESCRIPTION:
XS GIS Cut Line= 3
      1584726.69      6776059.76      1584966.30      6776227.83
      1585280.46      6776482.35
#Sta/Elev= 30
  4708.3 2072.30  4728.0 2071.51  4748.9 2068.71  4763.7 2070.29  4769.8 2068.42
  4778.5 2068.82  4784.6 2067.05  4799.4 2066.15  4805.5 2064.30  4814.2 2063.83
  4820.4 2062.04  4850.0 2058.02  4870.9 2052.68  4885.7 2041.08  4891.8 2040.39
  4900.5 2034.65  4906.6 2033.77  4913.9 2027.60  4921.5 2023.45  5007.5 2023.78
  5025.5 2022.59  5026.0 2022.09  5031.0 2022.59  5057.0 2023.42  5071.4 2028.05
  5077.8 2027.67  5085.8 2029.88  5192.4 2034.36  5242.4 2038.13  5405.3 2043.23
#Mann=3,-1,0
  4708.3    0.12       0  5025.5    0.07       0  5031.0    0.12       0
Bank Sta=5025.5,5031
Exp/Cntr=0.3,0.1

Type RM Length L Ch R = 1,14201,363,363,363
BEGIN DESCRIPTION:
Elm 01 74 14200.83
END DESCRIPTION:
XS GIS Cut Line= 3
      1584633.19      6776156.37      1584756.87      6776484.46
      1584932.17      6776803.89
#Sta/Elev= 30
  4651.5 2055.42  4694.9 2050.29  4706.7 2050.02  4755.3 2043.74  4770.8 2042.46
  4780.2 2042.78  4802.9 2039.78  4834.9 2031.77  4845.9 2027.18  4865.4 2021.56
  4870.8 2021.95  4888.4 2019.61  4909.7 2020.69  5014.8 2019.53  5015.3 2019.03
  5020.3 2019.53  5053.9 2021.06  5063.2 2020.31  5086.0 2022.11  5113.5 2026.22
  5120.2 2030.51  5129.6 2033.57  5135.3 2032.37  5143.0 2034.37  5200.7 2038.03
  5232.9 2038.69  5284.8 2041.34  5299.6 2042.61  5320.1 2043.55  5366.5 2047.79
#Mann=5,-1,0
  4651.5    0.12       0  5014.8    0.07       0  5020.3    0.12       0
  5284.8    0.05       0  5299.6    0.12       0
Bank Sta=5014.8,5020.3
Exp/Cntr=0.3,0.1

Type RM Length L Ch R = 1,13838,244,244,244
BEGIN DESCRIPTION:
Elm 01 74 13838.18
END DESCRIPTION:
XS GIS Cut Line= 3
      1584294.64      6776188.91      1584409.21      6776532.64
      1584566.77      6776910.26
#Sta/Elev= 30
  4639.7 2043.65  4655.6 2042.20  4660.9 2042.72  4687.2 2040.62  4724.1 2039.36
  4750.5 2036.98  4755.7 2037.35  4845.3 2032.31  4850.6 2032.59  4870.6 2031.41
  4877.0 2029.86  4882.2 2030.36  4891.7 2026.35  4902.3 2019.70  4908.6 2016.51
  4965.5 2017.21  4971.8 2016.46  5005.9 2015.76  5006.3 2015.26  5011.5 2015.76
  5032.5 2016.08  5050.9 2017.96  5056.3 2018.66  5062.0 2021.60  5085.5 2023.52
  5162.4 2026.57  5233.9 2032.23  5239.3 2031.75  5268.5 2033.09  5411.2 2041.43
#Mann=3,-1,0
  4639.7    0.12       0  5005.9    0.07       0  5011.5    0.12       0
Bank Sta=5005.9,5011.5
Exp/Cntr=0.3,0.1

Type RM Length L Ch R = 1,13594,306,306,306
BEGIN DESCRIPTION:
Elm 01 74 13593.86
END DESCRIPTION:
XS GIS Cut Line= 3
      1584094.59      6776415.12      1584202.25      6776644.32
      1584344.60      6776909.05
#Sta/Elev= 30
  4746.5 2025.37  4802.8 2024.44  4808.4 2024.94  4825.6 2024.30  4838.1 2024.71
  4876.8 2022.87  4916.8 2022.19  4937.5 2021.03  4950.7 2018.64  4959.6 2015.54
  4968.0 2013.88  4973.5 2013.48  4990.8 2015.42  4996.4 2014.13  5026.6 2014.45
  5037.6 2013.01  5038.1 2012.51  5042.8 2012.51  5043.2 2013.01  5049.3 2014.02
  5056.7 2013.84  5062.3 2014.90  5072.0 2017.83  5078.6 2022.19  5100.5 2024.23
  5144.3 2025.63  5196.9 2029.72  5219.6 2030.41  5232.0 2031.64  5300.3 2034.03
#Mann=4,-1,0
  4746.5    0.05       0  4916.8    0.12       0  5037.6    0.07       0
  5043.2    0.12       0
Bank Sta=5037.6,5043.2
Exp/Cntr=0.3,0.1

Type RM Length L Ch R = 1,13288,462,462,462
BEGIN DESCRIPTION:
Elm 01 74 13287.73
END DESCRIPTION:
XS GIS Cut Line= 3
      1583802.06      6776462.86      1583947.04      6776788.42
      1584053.82      6776990.68
#Sta/Elev= 30
  4644.1 2018.54  4726.4 2019.62  4734.6 2017.11  4740.1 2018.14  4757.8 2015.20
  4763.3 2016.88  4770.1 2014.21  4781.1 2011.56  4786.5 2012.27  4792.0 2010.42
  4800.2 2010.14  4800.6 2009.64  4805.8 2010.14  4848.0 2010.75  4908.2 2010.63
  4960.1 2011.98  4977.9 2010.83  4983.4 2012.69  5028.3 2011.54  5044.6 2014.52
  5050.3 2013.62  5056.5 2017.31  5066.6 2019.15  5094.3 2020.40  5116.3 2019.64
  5151.3 2021.88  5204.4 2024.52  5220.8 2027.16  5225.1 2029.67  5229.2 2029.67
#Mann=5,-1,0
  4644.1    0.05       0  4800.2    0.07       0  4805.8    0.05       0
  4848.0    0.12       0  5151.3    0.05       0
Bank Sta=4800.2,4805.8
Exp/Cntr=0.3,0.1

Type RM Length L Ch R = 1,12826,709,709,709
BEGIN DESCRIPTION:
Elm 01 74 12825.88
END DESCRIPTION:
XS GIS Cut Line= 4
      1583449.74      6776782.82      1583437.36      6776803.26
      1583558.01      6776890.36      1583871.11      6777229.41
#Sta/Elev= 30
  4826.8 2012.68  4848.0 2013.00  4860.1 2011.93  4873.0 2007.28  4881.5 2006.72
  4896.2 2007.81  4967.4 2007.77  5056.6 2006.33  5057.1 2005.83  5062.3 2006.33
  5102.2 2006.49  5144.5 2007.15  5172.9 2008.86  5179.7 2010.19  5208.0 2009.92
  5214.8 2010.53  5222.2 2012.71  5229.0 2012.23  5236.4 2014.60  5257.4 2016.00
  5284.9 2019.27  5293.1 2018.87  5328.2 2020.39  5335.6 2019.38  5342.4 2020.45
  5349.8 2019.32  5356.6 2020.88  5384.9 2022.37  5441.6 2024.88  5461.0 2024.88
#Mann=5,-1,0
  4826.8    0.05       0  5056.6    0.03       0  5062.3    0.05       0
  5102.2    0.12       0  5284.9    0.05       0
Bank Sta=5056.6,5062.3
Exp/Cntr=0.3,0.1

Type RM Length L Ch R = 1,12117,148,148,148
BEGIN DESCRIPTION:
Elm 01 74 12117.23
END DESCRIPTION:
XS GIS Cut Line= 3
      1583150.86      6776816.66      1583145.43      6777290.86
      1583163.87      6777653.16
#Sta/Elev= 30
  4528.4 2007.12  4539.7 2007.64  4559.7 2007.19  4611.2 2007.44  4645.2 2007.32
  4709.8 2007.39  4739.8 2008.21  4749.8 2007.76  4799.8 2008.85  4809.8 2008.47
  4819.8 2004.74  4829.8 2002.54  4879.8 2001.72  4899.8 2002.23  5006.9 2000.20
  5007.4 1999.70  5012.2 1999.70  5012.6 2000.20  5019.8 2000.82  5079.9 2002.00
  5099.9 2003.62  5119.9 2004.52  5140.0 2004.00  5200.0 2006.64  5280.1 2009.22
  5287.2 2010.10  5300.2 2010.44  5320.2 2011.80  5350.2 2011.89  5365.4 2012.52
#Mann=5,-1,0
  4528.4    0.05       0  4611.2    0.12       0  4645.2    0.05       0
  5006.9    0.05       0  5012.6    0.05       0
Bank Sta=5006.9,5012.6
Exp/Cntr=0.3,0.1

Type RM Length L Ch R = 1,11969,408,408,408
BEGIN DESCRIPTION:
Elm 01 74 11968.5
END DESCRIPTION:
XS GIS Cut Line= 3
      1582985.93      6776839.48      1582996.78      6777289.78
      1583015.23      6777660.89
#Sta/Elev= 30
  4551.3 2004.90  4579.8 2005.09  4589.8 2005.57  4639.8 2005.48  4669.9 2006.14
  4709.9 2006.17  4769.9 2006.95  4799.9 2006.80  4807.8 2006.36  4819.9 2006.32
  4829.9 2007.03  4839.9 2006.94  4849.9 2005.62  4859.9 2003.76  4879.9 1999.35
  4919.9 1998.25  4935.1 1998.26  4967.1 1997.62  4967.5 1997.12  4972.3 1997.12
  4972.8 1997.62  5033.2 1998.47  5110.1 1999.01  5170.2 2000.60  5190.2 2001.66
  5200.2 2001.66  5230.2 2003.55  5250.3 2004.15  5260.3 2004.86  5373.3 2009.07
#Mann=6,-1,0
  4551.3    0.12       0  4807.8    0.05       0  4935.1    0.12       0
  4967.1    0.07       0  4972.8    0.12       0  5033.2    0.05       0
Bank Sta=4967.1,4972.8
Exp/Cntr=0.3,0.1

Type RM Length L Ch R = 1,11561,443,443,443
BEGIN DESCRIPTION:
Elm 01 74 11560.73
END DESCRIPTION:
XS GIS Cut Line= 3
      1582592.50      6777060.04      1582604.65      6777337.81
      1582623.75      6777662.51
#Sta/Elev= 30
  4721.8 2000.60  4759.8 2000.54  4776.1 2000.19  4809.8 1999.19  4829.9 1998.99
  4839.9 1998.32  4849.9 1997.13  4874.3 1995.39  4889.1 1994.46  4894.1 1994.66
  4947.1 1991.88  4947.5 1991.38  4952.4 1991.38  4952.9 1991.88  4972.4 1992.26
  5002.4 1992.36  5010.0 1992.04  5030.1 1992.78  5050.1 1995.93  5060.1 1997.03
  5070.2 1997.52  5080.2 1998.66  5088.0 2000.22  5110.2 1999.52  5180.3 2000.51
  5220.4 1999.99  5230.4 2000.35  5250.5 2000.31  5310.6 2001.91  5325.1 2001.94
#Mann=6,-1,0
  4721.8    0.12       0  4776.1    0.05       0  4874.3    0.12       0
  4947.1    0.05       0  4952.9    0.12       0  4972.4    0.05       0
Bank Sta=4947.1,4952.9
Exp/Cntr=0.3,0.1

Type RM Length L Ch R = 1,11118,402,402,402
BEGIN DESCRIPTION:
Elm 01 74 11117.63
END DESCRIPTION:
XS GIS Cut Line= 3
      1582252.01      6776977.55      1582197.75      6777242.33
      1582135.91      6777551.52
#Sta/Elev= 30
  4731.2 1995.79  4772.5 1995.59  4794.5 1994.50  4833.7 1993.77  4839.8 1992.31
  4890.3 1990.57  4895.4 1990.89  4935.6 1989.14  4945.8 1989.40  4956.2 1989.94
  4976.6 1988.06  4986.0 1987.39  4991.1 1987.43  4996.7 1986.61  5007.3 1986.36
  5017.5 1985.30  5034.0 1982.70  5034.4 1982.20  5039.3 1982.20  5039.8 1982.70
  5042.0 1984.08  5048.1 1986.48  5068.5 1988.79  5093.0 1990.55  5099.0 1992.08
  5109.2 1992.54  5119.4 1992.89  5129.6 1992.47  5211.2 1993.71  5316.8 1993.00
#Mann=4,-1,0
  4731.2    0.12       0  4945.8    0.05       0  5034.0    0.03       0
  5039.8    0.05       0
Bank Sta=5034,5039.8
Exp/Cntr=0.3,0.1

Type RM Length L Ch R = 1,10716,166,166,166
BEGIN DESCRIPTION:
Elm 01 74 10716.42
END DESCRIPTION:
XS GIS Cut Line= 3
      1581822.32      6776773.58      1581827.74      6777139.24
      1581834.23      6777624.70
#Sta/Elev= 30
  4636.0 1988.69  4850.4 1989.09  4890.4 1988.59  4930.5 1989.67  4940.5 1989.27
  4960.5 1985.99  4980.5 1985.98  5001.7 1984.92  5010.5 1979.10  5017.6 1978.23
  5018.0 1977.73  5022.9 1977.73  5023.4 1978.23  5030.5 1983.97  5040.5 1985.28
  5070.5 1984.86  5100.5 1985.54  5110.5 1987.74  5130.5 1990.18  5140.5 1990.33
  5168.0 1988.78  5220.5 1988.27  5240.5 1989.24  5260.5 1986.77  5270.5 1986.76
  5280.5 1988.61  5320.5 1989.09  5430.5 1989.40  5450.5 1988.27  5487.2 1987.98
#Mann=3,-1,0
  4636.0    0.05       0  5017.6    0.03       0  5023.4    0.05       0
Bank Sta=5017.6,5023.4
Exp/Cntr=0.3,0.1

Type RM Length L Ch R = 1,10550,293,293,293
BEGIN DESCRIPTION:
Elm 01 74 10550.38
END DESCRIPTION:
XS GIS Cut Line= 3
      1581652.95      6777009.11      1581661.73      6777138.16
      1581685.60      6777630.73
#Sta/Elev= 30
  4871.3 1987.03  4890.2 1986.40  4900.3 1986.56  4910.3 1984.42  4920.3 1983.60
  4930.3 1984.12  4951.2 1984.36  4970.3 1984.10  4975.3 1984.43  4990.5 1979.02
  4998.1 1977.04  5007.6 1976.86  5008.0 1976.36  5012.9 1976.36  5013.4 1976.86
  5020.5 1977.22  5030.5 1981.11  5040.5 1984.11  5049.5 1985.44  5060.6 1986.58
  5168.6 1986.81  5173.6 1987.50  5180.7 1986.89  5200.7 1986.33  5290.8 1985.23
  5300.8 1984.74  5350.9 1984.11  5377.0 1984.85  5382.0 1984.68  5493.8 1985.48
#Mann=5,-1,0
  4871.3    0.05       0  4951.2    0.12       0  5007.6    0.07       0
  5013.4    0.12       0  5049.5    0.05       0
Bank Sta=5007.6,5013.4
Exp/Cntr=0.3,0.1

Type RM Length L Ch R = 1,10257,386,386,386
BEGIN DESCRIPTION:
Elm 01 74 10257.19
END DESCRIPTION:
XS GIS Cut Line= 3
      1581373.74      6777173.02      1581422.21      6777272.49
      1581564.38      6777577.43
#Sta/Elev= 30
  4889.5 1983.81  4902.2 1985.74  4907.8 1985.51  4917.3 1984.35  4939.5 1984.63
  4969.8 1983.72  4984.0 1981.76  4992.3 1978.81  4997.6 1974.16  5003.3 1973.95
  5003.8 1973.45  5008.7 1973.45  5009.2 1973.95  5015.2 1974.22  5020.7 1976.90
  5028.3 1978.62  5038.0 1979.64  5043.5 1982.05  5047.8 1982.06  5089.3 1982.09
  5094.8 1982.73  5105.5 1982.24  5117.7 1982.76  5140.5 1983.04  5157.9 1982.57
  5225.6 1982.73  5249.0 1982.83  5260.4 1983.25  5277.7 1982.95  5336.6 1983.27
#Mann=5,-1,0
  4889.5    0.05       0  5003.3    0.05       0  5009.2    0.05       0
  5047.8    0.12       0  5225.6    0.05       0
Bank Sta=5003.3,5009.2
Exp/Cntr=0.3,0.1

Type RM Length L Ch R = 1,9871,343,343,343
BEGIN DESCRIPTION:
Elm 01 74 9871.15
END DESCRIPTION:
XS GIS Cut Line= 4
      1580985.32      6777436.58      1581055.16      6777507.36
      1581253.67      6777595.39      1581571.34      6777752.07
#Sta/Elev= 30
  4681.7 1979.53  4696.7 1978.49  4767.4 1978.76  4802.8 1978.14  4871.5 1978.57
  4894.8 1980.31  4912.2 1979.24  4918.0 1980.73  4923.5 1981.02  4934.1 1980.58
  4946.8 1980.92  4964.6 1979.42  4977.9 1973.59  4990.4 1970.84  4990.9 1970.34
  4995.8 1970.34  4996.3 1970.84  4998.3 1975.02  5001.8 1975.02  5010.4 1978.88
  5016.0 1980.40  5022.1 1980.93  5077.8 1980.45  5150.7 1981.33  5178.7 1981.09
  5195.6 1981.66  5201.2 1981.16  5211.6 1981.87  5233.9 1981.69  5352.5 1984.06
#Mann=3,-1,0
  4681.7    0.05       0  4990.4    0.05       0  4996.3    0.05       0
Bank Sta=4990.4,4996.3
Exp/Cntr=0.3,0.1

Type RM Length L Ch R = 1,9528,262,262,262
BEGIN DESCRIPTION:
Elm 01 74 9528.24
END DESCRIPTION:
XS GIS Cut Line= 4
      1580770.49      6777563.76      1580961.79      6777798.35
      1581049.40      6777841.79      1581230.14      6777942.92
#Sta/Elev= 30
  4597.4 1977.65  4639.6 1976.19  4689.2 1975.59  4731.9 1976.15  4773.9 1975.96
  4809.3 1976.31  4831.3 1978.78  4837.8 1978.92  4845.7 1976.65  4860.1 1976.79
  4887.3 1977.83  4992.6 1978.13  4997.9 1977.89  5005.2 1976.64  5015.4 1973.65
  5021.2 1971.26  5024.3 1969.47  5024.7 1968.97  5029.7 1968.97  5030.2 1969.47
  5037.1 1970.18  5042.9 1974.16  5050.1 1977.38  5058.8 1978.79  5073.1 1979.24
  5096.0 1978.25  5102.2 1978.69  5161.6 1978.58  5176.2 1978.73  5205.0 1980.10
#Mann=3,-1,0
  4597.4    0.05       0  5024.3    0.05       0  5030.2    0.05       0
Bank Sta=5024.3,5030.2
Exp/Cntr=0.3,0.1

Type RM Length L Ch R = 1,9266,622,622,622
BEGIN DESCRIPTION:
Elm 01 74 9265.42
END DESCRIPTION:
XS GIS Cut Line= 5
      1580715.79      6777600.19      1580806.95      6777795.54
      1580825.88      6777938.36      1580838.20      6778105.43
      1580936.52      6778186.82
#Sta/Elev= 30
  4642.0 1975.91  4676.9 1975.72  4694.2 1974.96  4783.0 1975.35  4805.1 1975.96
  4819.6 1975.64  4827.2 1974.39  4836.9 1974.35  4878.0 1974.95  4956.4 1974.73
  4981.1 1975.18  4991.2 1972.84  4995.9 1968.77  4996.4 1968.27  5001.4 1968.27
  5001.9 1968.77  5011.3 1969.22  5021.3 1975.32  5041.4 1975.15  5057.0 1975.52
  5071.5 1976.57  5081.5 1978.08  5091.5 1977.98  5101.6 1976.67  5121.6 1975.24
  5131.6 1976.06  5190.6 1975.99  5204.0 1976.93  5275.2 1978.25  5296.8 1979.27
#Mann=3,-1,0
  4642.0    0.05       0  4995.9    0.05       0  5001.9    0.05       0
Bank Sta=4995.9,5001.9
Exp/Cntr=0.3,0.1

Type RM Length L Ch R = 1,8644,474,474,474
BEGIN DESCRIPTION:
Elm 01 74 8643.78
END DESCRIPTION:
XS GIS Cut Line= 3
      1580247.06      6777613.29      1580256.00      6777989.94
      1580266.42      6778300.71
#Sta/Elev= 30
  4625.9 1971.33  4690.6 1969.39  4730.6 1969.12  4790.7 1969.33  4810.7 1970.04
  4820.7 1971.68  4830.7 1969.70  4860.7 1970.48  4890.7 1970.18  4920.7 1971.07
  4940.7 1970.99  4970.7 1969.18  4980.7 1967.32  4987.7 1963.66  4988.2 1963.16
  4993.2 1963.16  4993.7 1963.66  5002.7 1964.01  5010.7 1967.09  5020.7 1969.10
  5030.7 1968.67  5048.3 1971.21  5050.7 1971.61  5090.8 1971.54  5123.4 1971.02
  5160.8 1971.22  5190.8 1970.81  5240.9 1971.54  5270.9 1972.33  5313.6 1974.82
#Mann=5,-1,0
  4625.9    0.05       0  4987.7    0.05       0  4993.7    0.05       0
  5048.3    0.12       0  5123.4    0.05       0
Bank Sta=4987.7,4993.7
Exp/Cntr=0.3,0.1

Type RM Length L Ch R = 1,8170,593,593,593
BEGIN DESCRIPTION:
Elm 01 74 8170.09
END DESCRIPTION:
XS GIS Cut Line= 4
      1579885.07      6777199.23      1579817.81      6777774.69
      1579825.44      6778040.29      1579838.74      6778294.15
#Sta/Elev= 30
  4157.0 1967.86  4165.8 1968.16  4195.9 1967.46  4206.1 1966.29  4316.9 1965.19
  4544.3 1965.36  4639.0 1964.94  4789.7 1965.97  4813.6 1967.81  4819.7 1966.74
  4849.7 1967.44  4882.3 1967.25  4919.8 1968.39  4929.8 1968.13  4939.8 1966.88
  4949.8 1966.53  4959.8 1964.12  4976.8 1961.65  4977.3 1961.15  4982.3 1961.15
  4982.8 1961.65  5002.1 1962.14  5009.8 1966.72  5025.3 1966.55  5049.9 1966.68
  5069.9 1968.32  5140.0 1968.05  5170.0 1968.57  5250.1 1970.92  5256.3 1971.66
#Mann=5,-1,0
  4157.0    0.05       0  4882.3    0.12       0  4976.8    0.07       0
  4982.8    0.12       0  5025.3    0.05       0
Bank Sta=4976.8,4982.8
Exp/Cntr=0.3,0.1

Type RM Length L Ch R = 1,7577,332,332,332
BEGIN DESCRIPTION:
Elm 01 74 7577
END DESCRIPTION:
XS GIS Cut Line= 4
      1579168.93      6776850.22      1579290.15      6777149.55
      1579314.71      6777790.17      1579322.88      6778300.67
#Sta/Elev= 30
  4037.1 1958.63  4088.2 1958.57  4093.6 1957.71  4117.8 1957.90  4120.1 1957.03
  4120.6 1956.53  4125.7 1956.53  4126.2 1957.03  4171.4 1957.56  4176.8 1958.13
  4230.4 1959.56  4254.5 1958.92  4598.7 1959.44  4778.8 1960.58  4968.9 1963.03
  4989.0 1957.87  4997.6 1960.01  5001.1 1960.01  5009.0 1962.12  5019.0 1963.55
  5039.0 1964.29  5049.0 1963.99  5069.0 1962.01  5099.0 1962.31  5119.0 1963.56
  5209.0 1963.92  5359.0 1966.19  5469.0 1965.68  5499.0 1964.16  5511.7 1964.62
#Mann=3,-1,0
  4037.1    0.05       0  4120.1    0.03       0  4126.2    0.05       0
Bank Sta=4120.1,4126.2
Exp/Cntr=0.3,0.1

Type RM Length L Ch R = 1,7245,547,547,547
BEGIN DESCRIPTION:
Elm 01 74 7244.93
END DESCRIPTION:
XS GIS Cut Line= 4
      1579030.91      6776456.95      1578970.48      6777238.32
      1578982.68      6777792.34      1578990.95      6778292.91
#Sta/Elev= 30
  3665.7 1957.17  3726.9 1955.44  3877.4 1952.82  3927.5 1953.84  3997.7 1952.97
  4064.8 1953.69  4128.1 1953.18  4709.1 1957.94  4749.2 1958.70  4759.2 1957.29
  4779.2 1958.26  4799.2 1958.12  4819.2 1958.88  4939.2 1959.18  4959.2 1960.00
  4969.2 1954.72  4976.2 1952.52  4976.7 1952.02  4981.8 1952.02  4982.3 1952.52
  5009.2 1954.12  5029.2 1960.09  5059.2 1959.32  5099.2 1959.50  5189.2 1960.94
  5229.3 1960.80  5289.3 1961.65  5399.3 1961.62  5489.3 1960.41  5504.2 1961.13
#Mann=3,-1,0
  3665.7    0.05       0  4976.2    0.03       0  4982.3    0.05       0
Bank Sta=4976.2,4982.3
Exp/Cntr=0.3,0.1

Type RM Length L Ch R = 1,6698,382,382,382
BEGIN DESCRIPTION:
Elm 01 74 6697.93
END DESCRIPTION:
XS GIS Cut Line= 4
      1579017.87      6776433.60      1578515.15      6777459.57
      1578450.34      6777744.05      1578429.56      6778103.86
#Sta/Elev= 30
  3568.6 1956.84  3588.3 1956.59  3610.8 1955.01  3662.6 1953.78  3790.8 1952.20
  3829.6 1952.73  3896.4 1952.00  4119.2 1952.24  4522.0 1953.71  4734.7 1953.16
  4750.5 1952.16  4777.7 1953.49  4853.1 1953.09  4883.9 1953.60  4894.1 1953.07
  4986.4 1954.11  5010.3 1953.24  5023.8 1948.64  5024.3 1948.14  5029.4 1948.14
  5029.9 1948.64  5036.9 1949.88  5046.9 1953.01  5056.9 1953.75  5147.1 1952.97
  5197.2 1953.13  5207.2 1953.91  5287.3 1953.75  5337.4 1955.20  5363.3 1954.66
#Mann=3,-1,0
  3568.6    0.05       0  5023.8    0.05       0  5029.9    0.05       0
Bank Sta=5023.8,5029.9
Exp/Cntr=0.3,0.1

Type RM Length L Ch R = 1,6316,544,544,544
BEGIN DESCRIPTION:
Elm 01 74 6315.8
END DESCRIPTION:
XS GIS Cut Line= 5
      1578853.83      6776350.22      1578130.58      6777332.58
      1578099.82      6777642.49      1578060.70      6777929.37
      1578073.45      6778068.13
#Sta/Elev= 30
  3470.3 1954.70  3560.9 1952.09  3682.0 1950.87  3776.1 1950.58  3876.3 1951.45
  3939.4 1950.29  4047.6 1950.69  4183.4 1949.96  4454.9 1950.14  4676.3 1949.20
  4755.9 1949.63  4766.0 1948.98  4794.2 1949.58  4926.8 1948.75  4987.1 1949.55
  5007.2 1949.30  5017.3 1947.19  5024.3 1947.02  5024.8 1946.52  5029.9 1946.52
  5030.4 1947.02  5037.5 1949.04  5047.6 1949.40  5168.7 1948.94  5223.3 1949.04
  5239.3 1949.65  5249.4 1949.16  5340.0 1949.86  5410.3 1949.66  5430.5 1950.86
#Mann=3,-1,0
  3470.3    0.05       0  5024.3    0.03       0  5030.4    0.05       0
Bank Sta=5024.3,5030.4
Exp/Cntr=0.3,0.1

Type RM Length L Ch R = 1,5772,296,296,296
BEGIN DESCRIPTION:
Elm 01 74 5771.7
END DESCRIPTION:
XS GIS Cut Line= 6
      1578082.13      6777081.99      1577918.33      6777313.04
      1577660.59      6777359.40      1577560.76      6777552.54
      1577808.43      6777812.40      1577842.54      6778031.65
#Sta/Elev= 30
  4393.4 1948.28  4751.1 1946.97  4846.8 1946.40  4862.9 1945.82  4923.9 1945.20
  4994.3 1945.76  5003.6 1944.19  5007.6 1944.19  5016.7 1945.73  5022.3 1946.14
  5028.4 1945.74  5061.7 1946.01  5067.3 1945.52  5095.3 1945.66  5112.2 1943.85
  5128.7 1943.71  5137.2 1942.73  5137.7 1942.23  5142.8 1942.23  5143.3 1942.73
  5177.2 1942.95  5247.6 1944.77  5318.4 1946.00  5431.6 1945.48  5525.5 1946.87
  5588.4 1947.07  5593.4 1947.57  5651.2 1947.99  5656.3 1948.43  5736.9 1948.44
#Mann=3,-1,0
  4393.4    0.05       0  5137.2    0.05       0  5143.3    0.05       0
Bank Sta=5137.2,5143.3
Exp/Cntr=0.3,0.1

Type RM Length L Ch R = 1,5476,78,78,78
BEGIN DESCRIPTION:
Elm 01 74 5476.2
END DESCRIPTION:
XS GIS Cut Line= 6
      1577901.48      6777246.55      1577356.77      6777339.87
      1577354.60      6777417.99      1577500.00      6777472.24
      1577495.66      6777561.22      1577775.64      6777852.05
#Sta/Elev= 30
  4423.5 1947.12  4581.7 1945.99  4713.2 1943.36  4733.1 1945.49  4738.2 1948.74
  4760.0 1950.43  4802.0 1947.05  4807.0 1949.05  4843.9 1947.66  4933.7 1949.73
  4938.8 1948.68  4953.0 1950.25  4979.2 1950.36  4994.7 1949.04  5083.8 1949.81
  5091.0 1950.84  5151.6 1948.41  5156.9 1949.56  5176.6 1948.67  5181.9 1950.06
  5212.2 1949.80  5220.1 1951.27  5236.1 1951.55  5241.9 1946.05  5251.9 1942.68
  5278.9 1941.72  5279.4 1941.22  5285.0 1941.72  5520.5 1945.65  5728.9 1946.46
#Mann=3,-1,0
  4423.5    0.05       0  5278.9    0.05       0  5285.0    0.05       0
Bank Sta=5278.9,5285
Exp/Cntr=0.3,0.1

Type RM Length L Ch R = 1,5398,192,192,192
BEGIN DESCRIPTION:
Elm 01 74 5397.65
END DESCRIPTION:
XS GIS Cut Line= 6
      1577814.66      6777172.77      1577365.45      6777218.34
      1577282.98      6777320.34      1577280.81      6777467.90
      1577400.17      6777543.86      1577738.70      6777901.92
#Sta/Elev= 30
  4420.6 1945.97  4530.8 1944.99  4561.0 1943.81  4671.5 1942.04  4691.6 1942.38
  4718.5 1941.75  4741.9 1942.12  4869.8 1939.64  4893.8 1939.89  4993.0 1939.17
  5007.9 1938.71  5008.4 1938.21  5013.5 1938.21  5014.0 1938.71  5070.9 1939.19
  5111.0 1940.17  5155.6 1939.91  5176.3 1940.54  5233.9 1940.44  5312.7 1941.57
  5319.9 1942.10  5461.5 1943.59  5496.7 1943.50  5588.6 1945.59  5602.7 1945.19
  5610.0 1945.65  5616.9 1945.40  5638.3 1945.83  5666.6 1945.34  5785.1 1946.44
#Mann=3,-1,0
  4420.6    0.05       0  5007.9    0.05       0  5014.0    0.05       0
Bank Sta=5007.9,5014
Exp/Cntr=0.3,0.1

Type RM Length L Ch R = 1,5206,538,538,538
BEGIN DESCRIPTION:
Elm 01 74 5205.81
END DESCRIPTION:
XS GIS Cut Line= 3
      1577263.32      6776661.93      1577103.59      6777283.48
      1577075.81      6777939.75
#Sta/Elev= 30
  4359.2 1939.45  4644.2 1937.84  4656.7 1937.39  4675.2 1937.79  4685.5 1937.34
  4716.5 1937.49  4757.8 1936.85  4773.8 1937.24  4850.1 1937.31  4855.3 1937.09
  4861.1 1935.76  4868.3 1933.06  4868.8 1932.56  4873.9 1932.56  4874.4 1933.06
  4881.7 1934.29  4890.9 1937.34  4936.8 1936.77  4954.0 1935.24  4972.3 1935.56
  4985.0 1934.52  5000.7 1936.72  5065.5 1937.08  5155.6 1938.47  5175.6 1938.12
  5235.7 1938.79  5326.5 1938.53  5505.9 1940.33  5626.0 1940.95  5657.8 1940.61
#Mann=3,-1,0
  4359.2    0.05       0  4868.3    0.03       0  4874.4    0.05       0
Bank Sta=4868.3,4874.4
Exp/Cntr=0.3,0.1

Type RM Length L Ch R = 1,4668,748,748,748
BEGIN DESCRIPTION:
Elm 01 74 4667.74
END DESCRIPTION:
XS GIS Cut Line= 3
      1576652.20      6776141.11      1576725.12      6776946.68
      1576676.51      6777887.66
#Sta/Elev= 30
  4198.2 1935.00  4282.6 1934.23  4287.6 1934.55  4295.5 1933.73  4325.6 1933.16
  4416.0 1932.87  4486.3 1933.06  4636.9 1935.36  4717.2 1934.03  4938.1 1934.20
  4946.7 1932.81  4951.7 1932.56  4958.2 1928.94  4968.2 1927.61  4988.3 1927.19
  5002.0 1925.87  5002.5 1925.37  5007.9 1925.37  5008.4 1925.87  5018.4 1926.54
  5028.4 1928.37  5078.5 1931.15  5088.5 1932.72  5104.9 1933.65  5348.8 1935.57
  5398.9 1936.45  5494.0 1936.38  5669.3 1938.01  5849.5 1938.50  5949.3 1938.04
#Mann=3,-1,0
  4198.2    0.05       0  5002.0    0.03       0  5008.4    0.05       0
Bank Sta=5002,5008.4
Exp/Cntr=0.3,0.1

Type RM Length L Ch R = 1,3920,608,608,608
BEGIN DESCRIPTION:
Elm 01 74 3920.43
END DESCRIPTION:
XS GIS Cut Line= 3
      1575989.01      6776116.80      1576023.73      6776991.82
      1576038.72      6778298.63
#Sta/Elev= 30
  4128.5 1925.96  4780.2 1925.55  4840.3 1926.00  4880.3 1927.07  4950.3 1927.14
  4980.4 1925.60  4996.6 1918.66  4997.1 1918.16  5002.5 1918.16  5003.0 1918.66
  5004.2 1918.66  5010.4 1922.89  5020.4 1926.31  5100.4 1926.02  5140.4 1925.06
  5280.4 1924.74  5360.4 1925.74  5490.4 1923.66  5548.1 1924.05  5553.1 1924.62
  5600.4 1924.49  5640.4 1925.77  5800.4 1925.04  6080.5 1921.33  6120.5 1922.81
  6200.5 1921.44  6240.5 1921.37  6270.5 1922.27  6290.5 1922.14  6311.1 1923.74
#Mann=3,-1,0
  4128.5    0.05       0  4996.6    0.03       0  5003.0    0.05       0
Bank Sta=4996.6,5003
Exp/Cntr=0.3,0.1

Type RM Length L Ch R = 1,3312,469,469,469
BEGIN DESCRIPTION:
Elm 01 74 3311.72
END DESCRIPTION:
XS GIS Cut Line= 3
      1575373.38      6776075.37      1575415.05      6776991.99
      1575444.09      6778293.60
#Sta/Elev= 30
  4086.8 1921.23  4730.1 1921.01  4760.1 1920.38  4800.2 1920.76  4900.3 1920.34
  4930.3 1920.56  4980.3 1922.05  4990.4 1918.68  4999.9 1916.29  5004.4 1916.29
  5010.4 1917.58  5020.4 1921.73  5050.4 1920.18  5080.4 1919.73  5290.4 1919.26
  5350.5 1919.82  5440.5 1919.25  5500.5 1920.11  5550.5 1919.12  5760.6 1918.48
  5900.6 1917.11  6110.7 1917.37  6200.7 1916.91  6237.5 1916.11  6238.0 1915.61
  6243.4 1915.61  6243.9 1916.11  6260.7 1916.83  6290.7 1916.69  6306.3 1917.60
#Mann=3,-1,0
  4086.8    0.05       0  6237.5    0.05       0  6243.9    0.05       0
Bank Sta=6237.5,6243.9
Exp/Cntr=0.3,0.1

Type RM Length L Ch R = 1,2843,468,468,468
BEGIN DESCRIPTION:
Elm 01 74 2842.86
END DESCRIPTION:
XS GIS Cut Line= 3
      1574908.10      6776033.69      1574946.30      6776995.46
      1575049.05      6778254.05
#Sta/Elev= 30
  4045.3 1919.44  4350.0 1918.49  4510.0 1917.18  4720.1 1916.59  4820.2 1917.26
  4910.3 1917.23  4960.3 1918.28  4980.3 1919.33  4990.4 1917.94  4997.2 1913.93
  4997.7 1913.43  5003.1 1913.43  5003.6 1913.93  5006.6 1916.78  5011.6 1916.78
  5020.4 1918.99  5049.4 1917.34  5100.7 1916.72  5191.0 1917.11  5411.7 1916.26
  5602.3 1916.55  5712.7 1915.99  5772.9 1916.64  5833.1 1915.42  6037.6 1914.30
  6073.9 1915.39  6104.0 1914.52  6159.3 1913.95  6244.5 1913.98  6270.6 1914.83
#Mann=3,-1,0
  4045.3    0.05       0  4997.2    0.05       0  5003.6    0.05       0
Bank Sta=4997.2,5003.6
Exp/Cntr=0.3,0.1
