--- Elm 01 78.prj (project) ---

Proj Title=Elm 01 78 Base Level Engineering
Current Plan=p01
Default Exp/Contr=0.3,0.1
English Units
Geom File=g01
Flow File=f01
Plan File=p01
Y Axis Title=Elevation
X Axis Title(PF)=Main Channel Distance
X Axis Title(XS)=Station
BEGIN DESCRIPTION:
Elm 01 78
END DESCRIPTION:
DSS Export Rating Curves= 0
DSS Export Rating Curve Sorted= 0
DSS Export Volume Flow Curves= 0
DXF OffsetX= 0
DXF OffsetY= 0
DXF ScaleX= 1
DXF ScaleY= 10

--- Elm 01 78.p01 (plan) ---

Plan Title=Multiple Run
Short Identifier=Multiple
Geom File=g01
Flow File=f01
Subcritical Flow
K Sum by GR= 0
Std Step Tol= 0.01
Critical Tol= 0.01
Num of Std Step Trials= 20
Max Error Tol= 0.3
Flow Tol Ratio= 0.001
Split Flow NTrial= 30
Split Flow Tol= 0.02
Split Flow Ratio= 0.02
Log Output Level= 0
Friction Slope Method= 1
Unsteady Friction Slope Method= 2
Unsteady Bridges Friction Slope Method= 1
Parabolic Critical Depth
Global Vel Dist=  1 , 1 , 1
Global Log Level= 0
CheckData=True
Encroach Param= -1, 0, 0, 0
BEGIN DESCRIPTION:
Multiple Run
END DESCRIPTION:

--- Elm 01 78.f01 (steady flow) ---

Flow Title=Multiple
Program Version=4.10
Number of Profiles= 7
Profile Names=10-year,25-year,50-year,1pct_min,100-year,1pct_plu,500-year
River Rch & RM=Elm 01 78,Reach-1         ,38593
     278     396     497     387     621     854     982
River Rch & RM=Elm 01 78,Reach-1         ,38045
     401     584     742     586     939    1290    1520
River Rch & RM=Elm 01 78,Reach-1         ,35864
     481     703     897     710    1140    1570    1850
River Rch & RM=Elm 01 78,Reach-1         ,30473
     553     807    1030     810    1300    1790    2100
River Rch & RM=Elm 01 78,Reach-1         ,29708
     553     807    1030     810    1300    1790    2100
River Rch & RM=Elm 01 78,Reach-1         ,19411
     688    1010    1300    1030    1650    2270    2710
River Rch & RM=Elm 01 78,Reach-1         ,17696
     705    1040    1330    1050    1680    2320    2750
River Rch & RM=Elm 01 78,Reach-1         ,16190
     912    1350    1740    1390    2220    3060    3670
River Rch & RM=Elm 01 78,Reach-1         ,12704
     912    1350    1740    1390    2220    3060    3670
River Rch & RM=Elm 01 78,Reach-1         ,8753
     985    1460    1890    1500    2410    3310    3970
River Rch & RM=Elm 01 78,Reach-1         ,5473
    1070    1580    2040    1630    2610    3590    4310
River Rch & RM=Elm 01 78,Reach-1         ,3121
    1070    1580    2040    1630    2610    3590    4310
Boundary for River Rch & Prof#=Elm 01 78,Reach-1         , 1
Up Type= 0
Dn Type= 3
Dn Slope=0.001
Boundary for River Rch & Prof#=Elm 01 78,Reach-1         , 2
Up Type= 0
Dn Type= 3
Dn Slope=0.001
Boundary for River Rch & Prof#=Elm 01 78,Reach-1         , 3
Up Type= 0
Dn Type= 3
Dn Slope=0.001
Boundary for River Rch & Prof#=Elm 01 78,Reach-1         , 4
Up Type= 0
Dn Type= 3
Dn Slope=0.001
Boundary for River Rch & Prof#=Elm 01 78,Reach-1         , 5
Up Type= 0
Dn Type= 3
Dn Slope=0.001
Boundary for River Rch & Prof#=Elm 01 78,Reach-1         , 6
Up Type= 0
Dn Type= 3
Dn Slope=0.001
Boundary for River Rch & Prof#=Elm 01 78,Reach-1         , 7
Up Type= 0
Dn Type= 3
Dn Slope=0.001
DSS Import GetInterval= 0
DSS Import GetPeak= 0
DSS Import FillOption= 0

--- Elm 01 78.g01 (geometry) ---

Geom Title=Existing Conditions

River Reach=Elm 01 78,Reach-1
Reach XY= 30
      1594405.00      6788838.00      1594598.77      6789330.19
      1595757.45      6789393.46      1596187.84      6790071.90
      1597199.75      6790643.44      1597060.07      6791140.29
      1598246.12      6792431.51      1597955.60      6792648.62
      1598004.02      6793877.74      1597156.53      6794493.88
      1597604.11      6795077.42      1596799.17      6797340.30
      1595641.68      6797901.37      1594557.97      6799046.34
      1594199.60      6800040.43      1592858.75      6801739.55
      1592803.80      6803177.50      1592055.54      6803772.46
      1592497.02      6803881.62      1592681.15      6804915.82
      1593053.55      6804641.04      1593452.00      6805030.28
      1592718.37      6805474.27      1592349.55      6806640.47
      1591618.23      6807074.33      1591006.87      6808293.69
      1591247.72      6808688.09      1590854.93      6810169.71
      1591255.00      6811388.00      1589305.00      6813038.00

Type RM Length L Ch R = 1,38593,290,290,290
BEGIN DESCRIPTION:
Elm 01 78 38418.69
END DESCRIPTION:
XS GIS Cut Line= 3
      1594142.04      6789018.61      1594418.63      6788851.42
      1594741.18      6788630.06
#Sta/Elev= 30
  4676.8 2031.09  4750.9 2031.38  4760.6 2030.55  4766.4 2031.14  4781.9 2030.10
  4861.5 2028.44  4890.6 2028.75  4941.1 2026.23  4984.1 2025.45  4993.4 2024.15
  5007.7 2023.79  5029.2 2024.93  5054.3 2023.16  5054.5 2022.66  5058.3 2023.16
  5065.1 2024.45  5071.2 2027.84  5092.6 2033.01  5121.9 2037.11  5157.8 2038.90
  5172.7 2038.40  5193.7 2039.93  5223.5 2039.66  5259.3 2041.18  5280.3 2043.63
  5331.1 2045.77  5359.4 2049.40  5366.9 2049.00  5373.0 2049.97  5391.2 2050.41
#Mann=3,-1,0
  4676.8    0.12       0  5054.3    0.07       0  5058.3    0.12       0
Bank Sta=5054.3,5058.3
Exp/Cntr=0.3,0.1

Type RM Length L Ch R = 1,38303,258,258,258
BEGIN DESCRIPTION:
Elm 01 78 38303.33
END DESCRIPTION:
XS GIS Cut Line= 3
      1593996.20      6789272.51      1594504.05      6789113.64
      1594851.32      6788873.92
#Sta/Elev= 30
  4467.2 2033.19  4598.2 2029.55  4603.5 2028.25  4644.1 2026.73  4663.2 2026.78
  4675.5 2027.93  4765.8 2025.49  4771.0 2024.36  4790.8 2024.07  4803.5 2021.88
  4830.7 2021.01  4853.6 2020.81  4874.6 2022.84  4906.1 2024.23  4987.8 2018.90
  4988.1 2018.40  4991.8 2018.90  5061.2 2020.70  5111.0 2025.10  5161.7 2027.89
  5248.2 2030.29  5298.9 2030.28  5340.8 2031.51  5349.6 2030.80  5355.7 2031.62
  5365.5 2030.76  5370.6 2031.48  5385.5 2030.19  5391.6 2030.97  5421.3 2030.81
#Mann=4,-1,0
  4467.2    0.12       0  4987.8    0.07       0  4991.8    0.12       0
  5365.5    0.05       0
Bank Sta=4987.8,4991.8
Exp/Cntr=0.3,0.1

Type RM Length L Ch R = 1,38045,511,511,511
BEGIN DESCRIPTION:
Elm 01 78 38044.83
END DESCRIPTION:
XS GIS Cut Line= 3
      1594281.39      6789568.08      1594586.08      6789318.07
      1595033.98      6788915.74
#Sta/Elev= 30
  4605.8 2031.03  4771.8 2024.77  4792.6 2022.66  4843.3 2022.03  4870.8 2018.99
  4942.6 2014.56  4985.6 2015.88  4989.9 2014.03  4990.2 2013.53  4994.3 2014.03
  5034.8 2017.27  5055.7 2021.37  5069.9 2020.78  5074.7 2021.69  5077.4 2022.20
  5084.1 2019.73  5091.6 2020.50  5098.3 2019.22  5126.7 2018.88  5224.1 2021.81
  5247.1 2023.94  5289.7 2023.89  5332.3 2025.93  5339.0 2027.28  5383.0 2028.79
  5402.5 2029.63  5473.5 2029.37  5481.0 2028.10  5487.7 2029.07  5602.0 2028.69
#Mann=6,-1,0
  4605.8    0.12       0  4989.9    0.07       0  4994.3    0.12       0
  5074.7    0.05       0  5224.1    0.12       0  5383.0    0.05       0
Bank Sta=4989.9,4994.3
Exp/Cntr=0.3,0.1

Type RM Length L Ch R = 1,37534,104,104,104
BEGIN DESCRIPTION:
Elm 01 78 37534.2
END DESCRIPTION:
XS GIS Cut Line= 4
      1594728.12      6789786.82      1595022.39      6789487.34
      1595064.06      6789413.12      1594963.79      6789177.44
#Sta/Elev= 30
  4579.1 2027.48  4795.3 2026.84  4837.7 2021.46  4844.7 2022.29  4851.8 2019.85
  4858.9 2020.00  4866.0 2017.77  4873.0 2018.06  4894.3 2013.31  4901.3 2013.36
  4908.4 2011.22  4915.4 2011.58  4922.6 2009.16  4929.6 2009.13  4950.9 2005.78
  4986.2 2005.09  4993.3 2003.67  5001.4 2003.92  5009.2 2002.20  5015.0 2002.93
  5030.9 2000.81  5050.3 2000.74  5050.7 2000.24  5054.8 2000.74  5089.3 2004.14
  5094.8 2003.28  5118.4 2007.50  5147.5 2010.24  5200.2 2017.82  5340.2 2021.84
#Mann=3,-1,0
  4579.1    0.05       0  5050.3    0.05       0  5054.8    0.05       0
Bank Sta=5050.3,5054.8
Exp/Cntr=0.3,0.1

Type RM Length L Ch R = 1,37430,76,76,76
BEGIN DESCRIPTION:
Elm 01 78 37430.25
END DESCRIPTION:
XS GIS Cut Line= 4
      1594837.48      6789823.30      1595121.35      6789506.87
      1595160.41      6789423.54      1595019.90      6789137.30
#Sta/Elev= 30
  4573.3 2025.41  4624.7 2024.35  4879.6 2023.25  4929.7 2021.69  4936.5 2020.58
  4943.2 2021.66  4997.4 2020.60  5084.7 2021.65  5089.9 2019.03  5096.8 2021.72
  5130.0 2020.79  5136.2 2019.59  5141.7 2020.43  5158.7 2019.51  5164.2 2020.34
  5174.6 2020.08  5181.1 2018.67  5186.7 2019.92  5203.6 2017.97  5209.2 2019.49
  5219.1 2018.90  5223.9 2016.74  5224.2 2016.24  5228.4 2016.74  5229.4 2017.34
  5231.7 2018.73  5248.6 2017.62  5302.4 2018.90  5406.0 2023.20  5409.3 2022.46
#Mann=5,-1,0
  4573.3    0.05       0  5223.9    0.05       0  5228.4    0.05       0
  5229.4    0.12       0  5302.4    0.05       0
Bank Sta=5223.9,5228.4
Exp/Cntr=0.3,0.1

Type RM Length L Ch R = 1,37354,230,230,230
BEGIN DESCRIPTION:
Elm 01 78 37353.86
END DESCRIPTION:
XS GIS Cut Line= 4
      1594901.31      6789901.39      1595187.76      6789538.12
      1595228.12      6789407.91      1595094.01      6789096.72
#Sta/Elev= 30
  4537.5 2022.98  4634.8 2022.35  4777.5 2023.14  4798.3 2022.36  4834.7 2023.35
  4876.9 2023.12  4885.0 2019.91  4891.4 2020.09  4898.4 2014.93  4905.8 2011.13
  4912.2 2010.34  4920.2 2007.34  4934.7 2003.73  4953.2 2003.36  4953.6 2002.86
  4957.4 2002.86  4957.7 2003.36  4969.9 2003.95  5031.7 2003.91  5039.2 2004.81
  5044.4 2003.91  5104.4 2008.88  5212.8 2011.00  5245.2 2015.96  5267.0 2013.43
  5277.9 2013.26  5306.8 2016.75  5321.5 2017.75  5347.6 2018.58  5475.3 2022.88
#Mann=5,-1,0
  4537.5    0.05       0  4953.2    0.05       0  4957.7    0.05       0
  5321.5    0.12       0  5347.6    0.05       0
Bank Sta=4953.2,4957.7
Exp/Cntr=0.3,0.1

Type RM Length L Ch R = 1,37124,324,324,324
BEGIN DESCRIPTION:
Elm 01 78 37124.44
END DESCRIPTION:
XS GIS Cut Line= 3
      1595375.47      6789956.57      1595402.82      6789496.89
      1595367.73      6789042.03
#Sta/Elev= 30
  4536.9 2011.86  4565.5 2013.06  4645.7 2013.68  4655.7 2014.48  4725.8 2013.28
  4775.9 2013.49  4795.9 2012.32  4826.0 2008.13  4836.0 2008.12  4856.0 2006.76
  4896.1 2005.19  4936.2 2001.85  4964.0 2001.34  4964.3 2000.84  4968.2 2000.84
  4968.5 2001.34  4984.8 2001.55  5037.7 2002.90  5096.6 2007.20  5116.6 2006.98
  5146.7 2008.12  5156.8 2008.91  5162.9 2010.02  5186.8 2011.60  5196.9 2011.28
  5206.9 2012.25  5306.0 2015.40  5357.3 2016.43  5397.5 2018.98  5453.6 2020.73
#Mann=5,-1,0
  4536.9    0.05       0  4964.0    0.07       0  4968.5    0.05       0
  4984.8    0.12       0  5306.0    0.05       0
Bank Sta=4964,4968.5
Exp/Cntr=0.3,0.1

Type RM Length L Ch R = 1,36800,195,195,195
BEGIN DESCRIPTION:
Elm 01 78 36800.47
END DESCRIPTION:
XS GIS Cut Line= 3
      1595561.69      6789567.08      1595677.56      6789390.03
      1595907.99      6789212.97
#Sta/Elev= 30
  4785.0 2005.66  4795.0 2006.40  4801.0 2005.12  4816.1 2006.20  4837.2 2004.42
  4852.3 2004.50  4867.4 2003.69  4939.3 2003.25  4966.8 2001.16  4981.9 1998.43
  5001.7 1997.97  5002.0 1997.47  5005.9 1997.47  5006.2 1997.97  5024.7 1998.50
  5039.2 1998.13  5074.6 1999.93  5089.1 1999.69  5109.9 2001.71  5118.1 2001.54
  5124.4 2002.36  5138.9 2002.14  5145.2 2003.35  5159.7 2004.90  5167.9 2005.23
  5195.1 2009.34  5203.3 2009.81  5238.6 2010.36  5253.1 2010.05  5287.2 2011.22
#Mann=3,-1,0
  4785.0    0.05       0  5001.7    0.05       0  5006.2    0.05       0
Bank Sta=5001.7,5006.2
Exp/Cntr=0.3,0.1

Type RM Length L Ch R = 1,36605,208,208,208
BEGIN DESCRIPTION:
Elm 01 78 36604.6
END DESCRIPTION:
XS GIS Cut Line= 3
      1595622.87      6789642.63      1595842.92      6789474.67
      1596081.14      6789274.00
#Sta/Elev= 30
  4723.9 2006.45  4821.6 2004.28  4865.0 2012.95  4900.5 2005.96  4906.8 2002.94
  4956.7 1996.70  4964.9 1994.28  4971.2 1994.89  4985.7 1991.60  4992.0 1993.35
  4998.9 1992.00  5006.6 1993.08  5014.4 1991.33  5020.9 1992.96  5028.7 1991.89
  5035.2 1993.45  5047.2 1991.20  5047.6 1990.70  5051.8 1991.20  5056.1 1993.02
  5063.8 1992.34  5070.4 1994.73  5078.1 1993.83  5084.7 1997.08  5092.4 1996.20
  5127.6 2003.70  5141.9 2001.31  5170.5 2006.11  5191.3 2007.32  5312.2 2010.66
#Mann=3,-1,0
  4723.9    0.05       0  5047.2    0.05       0  5051.8    0.05       0
Bank Sta=5047.2,5051.8
Exp/Cntr=0.3,0.1

Type RM Length L Ch R = 1,36397,136,136,136
BEGIN DESCRIPTION:
Elm 01 78 36396.81
END DESCRIPTION:
XS GIS Cut Line= 6
      1595637.16      6789705.14      1595825.99      6789663.47
      1595923.65      6789649.15      1595958.81      6789638.73
      1596023.91      6789612.69      1596137.19      6789304.09
#Sta/Elev= 30
  4669.8 2007.31  4817.5 2003.02  4822.6 2004.43  4841.7 2005.34  4863.2 2003.37
  4866.8 2006.19  4965.2 2005.79  4981.2 2001.83  4986.4 2005.07  4998.5 2004.91
  5012.3 2001.40  5017.7 2004.82  5036.5 2003.87  5041.9 2005.15  5059.1 2005.37
  5066.1 2004.22  5073.8 2005.10  5088.0 2003.84  5113.2 2003.93  5118.5 2001.95
  5143.6 2001.63  5146.7 1999.24  5147.0 1998.74  5151.3 1999.24  5168.8 1999.96
  5174.1 2002.29  5204.6 2004.66  5265.6 2005.60  5315.9 2008.03  5397.4 2009.90
#Mann=3,-1,0
  4669.8    0.05       0  5146.7    0.05       0  5151.3    0.05       0
Bank Sta=5146.7,5151.3
Exp/Cntr=0.3,0.1

Type RM Length L Ch R = 1,36261,397,397,397
BEGIN DESCRIPTION:
Elm 01 78 36260.54
END DESCRIPTION:
XS GIS Cut Line= 5
      1595667.13      6789765.03      1595941.88      6789723.37
      1596070.78      6789706.44      1596142.40      6789638.73
      1596221.82      6789334.07
#Sta/Elev= 30
  4590.4 2007.34  4719.7 2004.19  4736.1 2003.13  4765.8 2002.30  4799.8 2000.76
  4804.9 2001.03  4810.8 2000.21  4881.5 1997.29  4942.0 1995.97  4947.5 1995.37
  4952.5 1994.09  4982.4 1991.11  5004.9 1990.25  5005.2 1989.75  5009.1 1989.75
  5009.5 1990.25  5021.3 1990.70  5035.5 1993.19  5056.9 1994.59  5063.8 1995.72
  5106.0 1998.28  5125.2 2000.13  5130.4 2000.05  5149.3 2002.85  5165.7 2003.71
  5180.3 2003.53  5282.0 2006.07  5327.7 2008.35  5345.6 2008.12  5411.7 2009.80
#Mann=5,-1,0
  4590.4    0.05       0  4765.8    0.12       0  5004.9    0.07       0
  5009.5    0.12       0  5106.0    0.05       0
Bank Sta=5004.9,5009.5
Exp/Cntr=0.3,0.1

Type RM Length L Ch R = 1,35864,381,381,381
BEGIN DESCRIPTION:
Elm 01 78 35863.7
END DESCRIPTION:
XS GIS Cut Line= 3
      1595996.91      6790374.20      1596183.52      6790063.90
      1596396.18      6789634.24
#Sta/Elev= 30
  4640.4 2000.02  4717.6 2000.02  4739.3 1999.02  4766.5 1999.71  4811.0 1998.23
  4877.2 1998.23  4901.0 1997.33  4920.0 1996.24  4927.7 1995.26  4935.5 1992.82
  4941.3 1993.28  4972.4 1988.79  5002.5 1986.89  5009.1 1986.05  5013.5 1984.51
  5013.9 1984.01  5017.9 1984.01  5018.2 1984.51  5038.3 1987.70  5053.7 1988.33
  5083.2 1992.00  5128.0 1993.28  5150.5 1994.98  5209.6 1996.16  5262.6 1998.19
  5380.3 1999.75  5419.6 2001.47  5425.2 2000.80  5442.0 2002.01  5481.9 2002.04
#Mann=5,-1,0
  4640.4    0.05       0  4901.0    0.12       0  5013.5    0.07       0
  5018.2    0.12       0  5209.6    0.05       0
Bank Sta=5013.5,5018.2
Exp/Cntr=0.3,0.1

Type RM Length L Ch R = 1,35483,308,308,308
BEGIN DESCRIPTION:
Elm 01 78 35483.48
END DESCRIPTION:
XS GIS Cut Line= 3
      1596124.93      6790508.77      1596502.53      6790142.02
      1596743.26      6789792.86
#Sta/Elev= 30
  4468.0 1996.88  4539.2 1997.22  4574.7 1996.26  4610.0 1996.87  4645.4 1995.57
  4680.7 1995.69  4744.5 1994.12  4789.8 1991.40  4878.8 1988.41  4885.9 1987.39
  4892.9 1988.55  4907.0 1988.42  4921.2 1984.52  4975.4 1982.75  4975.7 1982.25
  4980.2 1982.75  4999.9 1983.03  5009.6 1984.47  5021.3 1985.53  5027.4 1987.20
  5042.3 1987.94  5057.2 1990.02  5114.0 1991.59  5149.8 1993.33  5164.7 1994.95
  5221.5 1996.09  5272.2 1998.95  5329.0 1999.21  5373.6 2001.38  5418.5 2002.06
#Mann=5,-1,0
  4468.0    0.05       0  4789.8    0.12       0  4975.4    0.07       0
  4980.2    0.12       0  5009.6    0.05       0
Bank Sta=4975.4,4980.2
Exp/Cntr=0.3,0.1

Type RM Length L Ch R = 1,35175,320,320,320
BEGIN DESCRIPTION:
Elm 01 78 35174.58
END DESCRIPTION:
XS GIS Cut Line= 3
      1596358.45      6790635.50      1596759.48      6790295.23
      1597004.30      6790040.00
#Sta/Elev= 30
  4475.3 1993.54  4527.7 1993.49  4549.5 1992.47  4562.8 1993.23  4584.8 1992.27
  4605.6 1992.64  4645.7 1990.90  4683.6 1987.97  4755.1 1984.44  4804.5 1985.02
  4917.6 1984.43  4953.9 1981.46  4960.4 1979.52  4979.8 1976.72  4980.2 1976.22
  4984.3 1976.22  4984.6 1976.72  5001.2 1977.82  5045.6 1988.10  5066.7 1990.31
  5121.8 1992.94  5137.4 1993.65  5165.7 1993.60  5179.9 1995.56  5201.3 1995.31
  5229.6 1996.21  5264.8 1999.07  5279.0 1998.67  5335.6 1999.64  5354.9 2000.97
#Mann=5,-1,0
  4475.3    0.05       0  4645.7    0.12       0  4979.8    0.07       0
  4984.6    0.12       0  5121.8    0.05       0
Bank Sta=4979.8,4984.6
Exp/Cntr=0.3,0.1

Type RM Length L Ch R = 1,34855,451,451,451
BEGIN DESCRIPTION:
Elm 01 78 34854.91
END DESCRIPTION:
XS GIS Cut Line= 3
      1596610.18      6790786.55      1596986.91      6790519.19
      1597318.48      6790253.59
#Sta/Elev= 30
  4538.0 1987.53  4597.5 1987.79  4612.3 1986.54  4618.4 1987.71  4648.0 1988.31
  4691.1 1987.59  4759.7 1984.64  4849.7 1981.98  4855.9 1981.16  4921.1 1978.22
  4942.0 1978.38  4985.4 1975.16  4994.3 1973.15  4994.6 1972.65  4999.1 1973.15
  5006.9 1973.21  5021.3 1977.97  5027.7 1978.37  5070.9 1978.52  5184.6 1982.60
  5248.6 1989.67  5263.0 1989.97  5269.4 1990.85  5277.4 1990.23  5298.2 1991.69
  5311.7 1991.71  5319.0 1992.74  5362.2 1993.30  5383.0 1995.31  5424.8 1995.75
#Mann=5,-1,0
  4538.0    0.05       0  4759.7    0.12       0  4994.3    0.07       0
  4999.1    0.12       0  5311.7    0.05       0
Bank Sta=4994.3,4999.1
Exp/Cntr=0.3,0.1

Type RM Length L Ch R = 1,34404,375,375,375
BEGIN DESCRIPTION:
Elm 01 78 34403.57
END DESCRIPTION:
XS GIS Cut Line= 3
      1596741.20      6790860.62      1597253.32      6790823.73
      1597701.32      6790773.96
#Sta/Elev= 30
  4485.8 1982.48  4509.7 1983.54  4549.8 1984.42  4588.4 1982.29  4593.4 1982.72
  4724.7 1978.55  4733.2 1979.03  4760.3 1977.33  4790.4 1976.96  4820.5 1973.95
  4850.5 1972.41  4942.9 1971.57  4950.8 1971.52  4970.9 1969.96  4988.5 1967.85
  4988.8 1967.35  4993.0 1967.35  4993.4 1967.85  4997.6 1969.35  5005.9 1969.32
  5011.0 1970.20  5047.1 1973.33  5061.3 1974.05  5091.5 1978.37  5101.6 1980.36
  5131.7 1982.69  5152.7 1983.61  5192.1 1985.12  5282.7 1987.24  5450.0 1987.72
#Mann=7,-1,0
  4485.8    0.05       0  4724.7    0.12       0  4942.9    0.05       0
  4988.5    0.05       0  4993.4    0.05       0  5047.1    0.12       0
  5152.7    0.05       0
Bank Sta=4988.5,4993.4
Exp/Cntr=0.3,0.1

Type RM Length L Ch R = 1,34029,266,266,266
BEGIN DESCRIPTION:
Elm 01 78 34029.24
END DESCRIPTION:
XS GIS Cut Line= 3
      1596350.55      6791168.79      1597053.66      6791125.38
      1597671.05      6790999.74
#Sta/Elev= 30
  4292.3 1988.01  4517.2 1985.68  4667.5 1982.02  4677.5 1981.58  4706.7 1977.04
  4727.6 1976.02  4787.7 1974.93  4797.7 1973.98  4817.8 1973.44  4847.8 1974.53
  4897.9 1973.52  4907.9 1972.44  4938.0 1965.05  4968.0 1963.65  5000.0 1963.80
  5003.5 1963.09  5003.9 1962.59  5008.1 1962.59  5008.5 1963.09  5018.5 1963.22
  5028.7 1964.95  5038.9 1965.76  5069.6 1966.44  5100.2 1968.16  5157.7 1974.05
  5294.1 1979.05  5334.9 1979.39  5360.1 1980.46  5396.1 1980.30  5626.8 1983.76
#Mann=3,-1,0
  4292.3    0.05       0  5003.5    0.05       0  5008.5    0.05       0
Bank Sta=5003.5,5008.5
Exp/Cntr=0.3,0.1

Type RM Length L Ch R = 1,33763,331,331,331
BEGIN DESCRIPTION:
Elm 01 78 33762.86
END DESCRIPTION:
XS GIS Cut Line= 3
      1596655.10      6791526.84      1597207.13      6791334.15
      1597637.68      6791205.68
#Sta/Elev= 30
  4413.8 1977.73  4515.4 1975.60  4520.7 1975.98  4625.5 1973.36  4639.6 1974.05
  4646.7 1972.87  4657.3 1972.35  4727.5 1971.61  4742.0 1972.07  4758.6 1971.30
  4789.6 1972.19  4869.1 1970.11  4882.8 1969.02  4939.6 1962.14  4976.0 1960.61
  4985.6 1959.11  4998.5 1958.64  4999.5 1958.02  4999.9 1957.52  5004.5 1958.02
  5027.6 1963.22  5040.4 1968.18  5048.5 1969.61  5073.5 1971.28  5111.9 1972.54
  5244.4 1974.29  5257.2 1975.05  5277.6 1975.02  5321.1 1977.35  5447.8 1979.44
#Mann=3,-1,0
  4413.8    0.05       0  4999.5    0.05       0  5004.5    0.05       0
Bank Sta=4999.5,5004.5
Exp/Cntr=0.3,0.1

Type RM Length L Ch R = 1,33432,355,355,355
BEGIN DESCRIPTION:
Elm 01 78 33432.4
END DESCRIPTION:
XS GIS Cut Line= 3
      1596913.76      6791943.51      1597401.58      6791592.83
      1597714.12      6791356.69
#Sta/Elev= 30
  4398.8 1978.65  4619.1 1972.97  4690.3 1970.14  4740.7 1965.96  4782.4 1959.75
  4819.1 1959.93  4826.6 1960.47  4832.8 1963.97  4847.5 1966.29  4883.1 1966.86
  4897.8 1964.53  4912.5 1957.76  4918.7 1956.73  4948.1 1955.69  4969.0 1956.33
  4975.1 1955.02  4975.5 1954.52  4980.1 1955.02  4998.5 1956.88  5041.5 1958.48
  5077.5 1961.51  5091.6 1963.67  5112.9 1962.13  5127.5 1962.97  5148.3 1964.82
  5154.6 1966.68  5169.1 1966.72  5254.5 1973.46  5368.9 1978.62  5391.3 1978.50
#Mann=3,-1,0
  4398.8    0.05       0  4975.1    0.05       0  4980.1    0.05       0
Bank Sta=4975.1,4980.1
Exp/Cntr=0.3,0.1

Type RM Length L Ch R = 1,33077,415,415,415
BEGIN DESCRIPTION:
Elm 01 78 33077.19
END DESCRIPTION:
XS GIS Cut Line= 3
      1597428.48      6792167.51      1597606.87      6791843.27
      1597789.00      6791442.59
#Sta/Elev= 30
  4631.1 1970.59  4700.6 1968.41  4716.7 1969.58  4722.4 1968.22  4813.2 1965.02
  4857.8 1961.91  4870.2 1959.34  4923.1 1952.71  4950.6 1952.17  4972.9 1952.62
  4982.8 1952.09  4992.9 1949.60  4993.3 1949.10  4997.9 1949.10  4998.3 1949.60
  5010.6 1951.17  5039.9 1953.30  5072.9 1953.42  5131.4 1955.83  5138.8 1957.22
  5171.7 1960.77  5183.1 1962.80  5215.7 1964.26  5275.3 1965.55  5314.5 1968.89
  5344.5 1973.66  5390.7 1976.52  5396.2 1976.25  5419.2 1977.67  5441.3 1978.04
#Mann=3,-1,0
  4631.1    0.05       0  4992.9    0.05       0  4998.3    0.05       0
Bank Sta=4992.9,4998.3
Exp/Cntr=0.3,0.1

Type RM Length L Ch R = 1,32662,503,503,503
BEGIN DESCRIPTION:
Elm 01 78 32662.36
END DESCRIPTION:
XS GIS Cut Line= 3
      1597583.18      6792234.13      1597947.80      6792044.87
      1598245.46      6791641.65
#Sta/Elev= 30
  4587.0 1967.70  4608.6 1968.61  4622.9 1966.87  4724.8 1964.16  4807.6 1964.03
  4814.4 1963.38  4824.1 1960.84  4836.9 1954.69  4846.2 1952.40  4851.9 1949.64
  4868.4 1948.54  4899.4 1949.23  4949.6 1948.82  4969.4 1945.43  4969.8 1944.93
  4974.9 1945.43  4979.0 1946.93  5007.0 1950.73  5086.4 1951.83  5136.5 1953.71
  5201.3 1954.07  5279.8 1959.47  5328.0 1960.94  5422.6 1964.95  5437.2 1964.82
  5451.9 1966.29  5458.1 1968.14  5472.7 1967.49  5478.9 1969.91  5499.0 1970.29
#Mann=5,-1,0
  4587.0    0.05       0  4899.4    0.12       0  4969.4    0.07       0
  4974.9    0.12       0  5328.0    0.05       0
Bank Sta=4969.4,4974.9
Exp/Cntr=0.3,0.1

Type RM Length L Ch R = 1,32159,204,204,204
BEGIN DESCRIPTION:
Elm 01 78 32158.63
END DESCRIPTION:
XS GIS Cut Line= 3
      1597647.43      6792234.10      1598246.41      6792433.76
      1598870.72      6792430.29
#Sta/Elev= 30
  4368.6 1966.97  4482.0 1964.51  4597.9 1959.07  4615.9 1957.33  4621.2 1957.73
  4684.4 1953.11  4724.4 1948.26  4769.7 1945.39  4810.9 1944.00  4837.3 1944.64
  4874.2 1943.76  4893.1 1944.96  4945.8 1944.72  4977.4 1943.56  4995.4 1942.21
  4996.0 1941.14  4996.4 1940.64  5001.5 1941.14  5008.6 1944.41  5093.6 1943.28
  5100.7 1943.37  5128.6 1943.16  5148.6 1944.19  5178.6 1948.14  5208.6 1950.25
  5366.3 1954.01  5408.6 1956.09  5448.6 1956.77  5488.6 1958.68  5624.3 1958.95
#Mann=7,-1,0
  4368.6    0.05       0  4769.7    0.12       0  4996.0    0.07       0
  5001.5    0.12       0  5093.6    0.05       0  5100.7    0.12       0
  5366.3    0.05       0
Bank Sta=4996,5001.5
Exp/Cntr=0.3,0.1

Type RM Length L Ch R = 1,31955,60,60,60
BEGIN DESCRIPTION:
Elm 01 78 31955.01
END DESCRIPTION:
XS GIS Cut Line= 6
      1597637.02      6792334.80      1598067.59      6792447.65
      1598079.75      6792517.09      1598124.89      6792560.50
      1598248.15      6792569.18      1598857.57      6792504.94
#Sta/Elev= 30
  4487.2 1966.96  4560.8 1963.84  4682.0 1954.75  4717.2 1954.93  4733.2 1956.68
  4784.9 1952.71  4826.3 1945.74  4857.3 1943.88  4919.3 1942.75  4942.0 1943.79
  4953.0 1947.12  4963.1 1947.77  5000.7 1946.46  5032.7 1947.48  5100.9 1946.60
  5105.9 1948.16  5195.9 1948.98  5205.9 1948.43  5226.1 1943.39  5273.5 1941.90
  5274.0 1941.40  5279.1 1941.90  5342.5 1947.00  5488.4 1949.32  5539.8 1951.19
  5598.1 1954.93  5631.4 1954.49  5668.5 1958.25  5718.8 1956.50  5801.8 1958.79
#Mann=7,-1,0
  4487.2    0.05       0  4857.3    0.12       0  5032.7    0.05       0
  5273.5    0.07       0  5279.1    0.05       0  5488.4    0.12       0
  5539.8    0.05       0
Bank Sta=5273.5,5279.1
Exp/Cntr=0.3,0.1

Type RM Length L Ch R = 1,31895,471,471,471
BEGIN DESCRIPTION:
Elm 01 78 31894.89
END DESCRIPTION:
XS GIS Cut Line= 5
      1597536.35      6792425.08      1598038.08      6792557.02
      1598133.57      6792638.62      1598321.07      6792633.41
      1598888.78      6792591.75
#Sta/Elev= 30
  4482.8 1967.62  4584.8 1964.56  4615.8 1962.63  4636.8 1960.07  4666.8 1959.76
  4719.2 1954.99  4752.6 1953.26  4787.8 1949.42  4822.6 1948.35  4863.3 1943.77
  4868.5 1944.54  4884.7 1941.54  4904.9 1940.60  4915.7 1940.48  4936.4 1942.59
  4946.4 1938.86  4946.8 1938.36  4952.0 1938.86  4957.0 1940.06  4977.7 1941.19
  5008.6 1941.63  5288.7 1941.78  5378.9 1945.98  5417.0 1946.70  5483.3 1947.67
  5569.4 1948.99  5659.6 1954.66  5689.7 1953.61  5749.9 1956.42  5884.0 1957.20
#Mann=7,-1,0
  4482.8    0.05       0  4904.9    0.12       0  4946.4    0.07       0
  4952.0    0.12       0  5008.6    0.05       0  5417.0    0.12       0
  5483.3    0.05       0
Bank Sta=4946.4,4952
Exp/Cntr=0.3,0.1

Type RM Length L Ch R = 1,31424,253,253,253
BEGIN DESCRIPTION:
Elm 01 78 31424.14
END DESCRIPTION:
XS GIS Cut Line= 3
      1597398.81      6792991.98      1598001.19      6792979.83
      1598730.19      6792936.43
#Sta/Elev= 30
  4393.5 1971.26  4459.7 1969.16  4499.7 1966.09  4539.7 1960.94  4569.7 1954.66
  4589.7 1951.59  4621.2 1950.26  4659.7 1946.22  4749.8 1941.57  4789.8 1940.89
  4799.8 1939.67  4809.8 1937.22  4889.8 1935.65  4906.9 1934.06  4907.4 1933.56
  4912.6 1934.06  4919.8 1936.33  4929.8 1937.61  4989.8 1937.29  4995.4 1935.42
  5009.8 1934.44  5018.9 1936.46  5234.1 1937.10  5282.2 1937.56  5300.4 1939.03
  5340.4 1940.19  5420.0 1947.91  5590.9 1953.17  5671.0 1952.82  5726.3 1954.32
#Mann=7,-1,0
  4393.5    0.05       0  4621.2    0.12       0  4906.9    0.07       0
  4912.6    0.12       0  5018.9    0.05       0  5234.1    0.12       0
  5420.0    0.05       0
Bank Sta=4906.9,4912.6
Exp/Cntr=0.3,0.1

Type RM Length L Ch R = 1,31171,434,434,434
BEGIN DESCRIPTION:
Elm 01 78 31170.51
END DESCRIPTION:
XS GIS Cut Line= 3
      1597278.98      6793262.81      1598004.66      6793233.30
      1598747.74      6793158.64
#Sta/Elev= 30
  4272.9 1971.48  4319.0 1969.80  4359.0 1966.65  4449.1 1953.06  4549.7 1944.74
  4599.2 1941.71  4619.2 1939.66  4689.3 1936.24  4817.0 1933.57  4869.4 1934.30
  4879.4 1932.67  4886.6 1932.62  4887.0 1932.12  4892.3 1932.62  4916.1 1934.09
  4959.5 1933.35  5003.3 1933.96  5009.6 1932.83  5029.7 1933.91  5150.3 1935.85
  5160.3 1937.04  5180.4 1936.97  5240.7 1939.01  5304.2 1943.00  5341.2 1946.42
  5404.4 1949.85  5414.4 1949.72  5562.3 1951.10  5582.4 1949.92  5746.0 1950.23
#Mann=7,-1,0
  4272.9    0.05       0  4549.7    0.12       0  4817.0    0.05       0
  4886.6    0.07       0  4892.3    0.05       0  4916.1    0.12       0
  5414.4    0.05       0
Bank Sta=4886.6,4892.3
Exp/Cntr=0.3,0.1

Type RM Length L Ch R = 1,30737,264,264,264
BEGIN DESCRIPTION:
Elm 01 78 30737.31
END DESCRIPTION:
XS GIS Cut Line= 3
      1597189.17      6793445.27      1597956.57      6793605.00
      1598727.40      6793559.86
#Sta/Elev= 30
  4216.9 1966.44  4301.7 1961.98  4335.2 1958.40  4365.9 1953.12  4376.1 1952.32
  4452.3 1949.12  4468.0 1948.68  4529.3 1943.61  4660.3 1936.93  4754.0 1932.45
  4856.1 1930.17  4927.6 1931.52  4983.2 1931.18  4992.5 1930.58  5006.3 1927.17
  5006.8 1926.67  5012.0 1927.17  5029.2 1929.98  5034.6 1930.13  5039.6 1928.93
  5049.3 1930.41  5099.3 1932.30  5139.4 1935.82  5253.3 1940.56  5279.7 1942.32
  5289.7 1941.86  5389.8 1944.73  5551.6 1947.25  5590.2 1945.32  5772.9 1945.28
#Mann=7,-1,0
  4216.9    0.05       0  4452.3    0.12       0  4660.3    0.05       0
  4983.2    0.12       0  5006.3    0.07       0  5012.0    0.12       0
  5253.3    0.05       0
Bank Sta=5006.3,5012
Exp/Cntr=0.3,0.1

Type RM Length L Ch R = 1,30473,510,510,510
BEGIN DESCRIPTION:
Elm 01 78 30472.64
END DESCRIPTION:
XS GIS Cut Line= 4
      1596329.18      6793706.21      1597374.84      6793718.49
      1598006.66      6793853.78      1598671.42      6793868.94
#Sta/Elev= 30
  3309.4 1968.56  3395.2 1967.45  3586.4 1957.05  3605.2 1952.79  3635.2 1939.81
  3645.2 1939.45  3695.2 1937.73  3725.2 1941.36  3825.3 1941.09  3905.3 1938.74
  3975.3 1942.77  4023.9 1941.32  4065.3 1938.78  4105.3 1938.96  4155.3 1942.94
  4185.3 1940.22  4295.3 1946.29  4508.7 1939.25  4651.9 1930.03  4815.5 1928.63
  4938.2 1931.32  4988.3 1927.69  5006.8 1925.71  5007.2 1925.21  5012.5 1925.71
  5029.6 1932.59  5039.6 1934.24  5294.9 1940.91  5469.7 1942.86  5666.2 1941.56
#Mann=7,-1,0
  3309.4    0.05       0  3586.4    0.12       0  4023.9    0.05       0
  4988.3    0.12       0  5006.8    0.07       0  5012.5    0.12       0
  5294.9    0.05       0
Bank Sta=5006.8,5012.5
Exp/Cntr=0.3,0.1

Type RM Length L Ch R = 1,29963,255,255,255
BEGIN DESCRIPTION:
Elm 01 78 29962.97
END DESCRIPTION:
XS GIS Cut Line= 4
      1596602.62      6793953.61      1597403.36      6793888.51
      1597583.48      6793962.29      1598505.83      6794072.97
#Sta/Elev= 30
  4004.7 1960.09  4216.2 1952.60  4247.9 1950.28  4284.1 1942.49  4368.3 1933.10
  4382.9 1934.64  4418.4 1932.81  4649.2 1933.14  4659.2 1933.34  4679.3 1937.98
  4713.8 1938.31  4822.2 1938.95  4841.6 1938.53  4863.9 1935.50  4871.0 1935.65
  4876.4 1938.21  4895.0 1938.13  4899.4 1936.53  4917.9 1935.21  4929.8 1930.33
  4948.4 1926.84  4953.8 1924.44  4997.9 1923.56  4998.4 1923.06  5003.7 1923.56
  5091.2 1927.36  5222.5 1927.75  5356.8 1928.18  5507.5 1932.88  5931.7 1939.68
#Mann=9,-1,0
  4004.7    0.05       0  4216.2    0.12       0  4284.1    0.05       0
  4713.8    0.12       0  4822.2    0.05       0  4899.4    0.12       0
  4997.9    0.07       0  5003.7    0.12       0  5222.5    0.05       0
Bank Sta=4997.9,5003.7
Exp/Cntr=0.3,0.1

Type RM Length L Ch R = 1,29708,482,482,482
BEGIN DESCRIPTION:
Elm 01 78 29870.88
END DESCRIPTION:
XS GIS Cut Line= 3
      1596656.80      6794120.71      1597404.90      6794119.81
      1598490.30      6794185.80
#Sta/Elev= 30
  4251.9 1957.06  4300.1 1956.15  4362.0 1953.20  4400.1 1952.22  4440.1 1949.09
  4450.1 1949.99  4510.1 1947.60  4570.1 1943.03  4660.1 1939.49  4700.1 1940.24
  4720.1 1935.73  4730.1 1931.89  4780.1 1926.96  4810.1 1925.17  4887.3 1924.40
  5007.0 1922.66  5007.5 1922.16  5013.2 1922.66  5053.9 1923.48  5100.3 1926.02
  5160.4 1924.90  5340.7 1926.80  5393.2 1926.22  5440.9 1924.86  5460.9 1926.10
  5531.1 1925.65  5691.4 1931.76  5741.5 1931.30  5931.8 1936.40  6087.4 1939.31
#Mann=6,-1,0
  4251.9    0.12       0  4362.0    0.05       0  4887.3    0.12       0
  5007.0    0.07       0  5013.2    0.12       0  5393.2    0.05       0
Bank Sta=5007,5013.2
Exp/Cntr=0.3,0.1

Type RM Length L Ch R = 1,29226,540,540,540
BEGIN DESCRIPTION:
Elm 01 78 29439.88
END DESCRIPTION:
XS GIS Cut Line= 3
      1596209.75      6794522.19      1597156.53      6794493.88
      1598768.40      6794530.87
#Sta/Elev= 30
  4052.8 1958.08  4178.1 1957.15  4318.2 1953.31  4356.7 1951.27  4424.8 1942.17
  4468.2 1935.72  4508.3 1932.98  4528.3 1933.58  4558.3 1932.52  4588.3 1934.01
  4680.8 1932.34  4728.4 1932.65  4799.7 1930.80  4968.5 1927.54  4978.5 1926.42
  4996.7 1920.99  5008.5 1918.78  5018.5 1919.98  5048.5 1920.35  5208.5 1919.65
  5258.5 1922.47  5415.4 1918.77  5415.9 1918.27  5421.7 1918.77  5630.8 1921.12
  5948.7 1927.78  6078.8 1929.36  6228.8 1933.51  6388.8 1935.37  6612.3 1934.52
#Mann=7,-1,0
  4052.8    0.05       0  4424.8    0.12       0  4680.8    0.05       0
  4799.7    0.12       0  5415.4    0.07       0  5421.7    0.12       0
  5630.8    0.05       0
Bank Sta=5415.4,5421.7
Exp/Cntr=0.3,0.1

Type RM Length L Ch R = 1,28686,776,776,776
BEGIN DESCRIPTION:
Elm 01 78 28686.25
END DESCRIPTION:
XS GIS Cut Line= 3
      1596602.97      6794907.46      1597460.65      6794829.33
      1598461.24      6794642.05
#Sta/Elev= 30
  4142.0 1952.94  4244.5 1951.49  4274.6 1948.31  4300.6 1942.44  4305.6 1943.31
  4334.8 1937.30  4375.0 1932.38  4455.3 1927.48  4535.7 1919.59  4589.4 1918.95
  4696.3 1918.19  4825.0 1921.48  4907.2 1922.65  4947.4 1918.81  4981.9 1917.45
  4997.6 1916.89  5002.9 1914.79  5008.0 1914.79  5014.7 1911.79  5015.2 1911.29
  5021.0 1911.79  5048.4 1917.00  5078.9 1918.42  5160.3 1917.16  5330.4 1919.00
  5366.3 1919.58  5384.1 1921.27  5692.1 1926.91  5760.5 1926.84  6021.2 1933.36
#Mann=7,-1,0
  4142.0    0.05       0  4589.4    0.12       0  4825.0    0.05       0
  4981.9    0.12       0  5014.7    0.07       0  5021.0    0.12       0
  5330.4    0.05       0
Bank Sta=5014.7,5021
Exp/Cntr=0.3,0.1

Type RM Length L Ch R = 1,27910,336,336,336
BEGIN DESCRIPTION:
Elm 01 78 27909.68
END DESCRIPTION:
XS GIS Cut Line= 3
      1596757.57      6795428.29      1597304.40      6795365.79
      1598380.37      6795154.07
#Sta/Elev= 30
  4449.8 1950.39  4494.4 1950.93  4499.5 1949.16  4593.2 1949.95  4596.2 1950.11
  4618.3 1948.87  4648.5 1943.11  4668.1 1941.72  4673.1 1939.17  4688.8 1935.22
  4729.0 1921.64  4749.2 1916.31  4802.9 1912.90  4880.0 1911.74  4950.5 1913.14
  4994.7 1907.26  4995.2 1906.76  5001.2 1907.26  5031.4 1911.93  5082.3 1913.48
  5277.3 1914.29  5357.5 1916.65  5484.8 1917.34  5561.4 1917.36  5580.5 1918.94
  5673.3 1920.37  5816.1 1923.94  5899.0 1927.30  6056.9 1930.59  6096.8 1929.61
#Mann=9,-1,0
  4449.8    0.05       0  4593.2    0.12       0  4596.2    0.05       0
  4802.9    0.12       0  4994.7    0.07       0  5001.2    0.12       0
  5484.8    0.05       0  5673.3    0.12       0  6056.9    0.05       0
Bank Sta=4994.7,5001.2
Exp/Cntr=0.3,0.1

Type RM Length L Ch R = 1,27574,649,649,649
BEGIN DESCRIPTION:
Elm 01 78 27574.26
END DESCRIPTION:
XS GIS Cut Line= 3
      1596577.38      6795719.78      1597306.54      6795674.21
      1598387.24      6795567.88
#Sta/Elev= 30
  4269.1 1962.37  4382.0 1958.23  4467.1 1954.84  4557.0 1954.17  4748.9 1954.79
  4807.8 1954.09  4817.8 1952.35  4853.4 1935.27  4855.8 1933.97  4860.8 1934.26
  4887.9 1921.10  4918.0 1911.52  4938.0 1909.08  4968.1 1910.50  5004.3 1905.12
  5004.8 1904.62  5010.9 1905.12  5012.6 1906.91  5018.2 1905.46  5038.3 1910.29
  5215.2 1910.63  5473.6 1914.59  5550.8 1913.74  5570.9 1916.44  5591.0 1916.99
  5620.5 1915.62  5762.7 1922.48  5821.7 1923.65  6030.7 1927.82  6085.6 1926.82
#Mann=10,-1,0
  4269.1    0.12       0  4382.0    0.05       0  4557.0    0.12       0
  4748.9    0.05       0  4853.4    0.12       0  5004.3    0.07       0
  5010.9    0.12       0  5473.6    0.05       0  5762.7    0.12       0
  5821.7    0.05       0
Bank Sta=5004.3,5010.9
Exp/Cntr=0.3,0.1

Type RM Length L Ch R = 1,26925,784,784,784
BEGIN DESCRIPTION:
Elm 01 78 27047.52
END DESCRIPTION:
XS GIS Cut Line= 3
      1596579.72      6795923.77      1597304.17      6796138.84
      1598097.88      6796418.39
#Sta/Elev= 30
  4244.3 1956.94  4348.0 1951.03  4406.3 1948.87  4419.6 1947.30  4435.5 1942.16
  4447.6 1937.20  4452.8 1936.96  4458.4 1933.21  4486.0 1923.48  4491.3 1923.29
  4519.3 1916.52  4557.7 1911.53  4590.9 1908.94  4772.6 1905.77  4844.4 1907.35
  4982.3 1906.52  4990.4 1906.32  4997.8 1903.60  5014.7 1902.02  5018.8 1900.60
  5019.3 1900.10  5025.4 1900.60  5064.5 1907.12  5244.7 1905.80  5282.6 1907.59
  5525.0 1908.57  5555.9 1909.40  5563.2 1910.71  5648.8 1910.93  5841.5 1917.52
#Mann=5,-1,0
  4244.3    0.05       0  4435.5    0.12       0  5018.8    0.07       0
  5025.4    0.12       0  5563.2    0.05       0
Bank Sta=5018.8,5025.4
Exp/Cntr=0.3,0.1

Type RM Length L Ch R = 1,26141,427,427,427
BEGIN DESCRIPTION:
Elm 01 78 26140.98
END DESCRIPTION:
XS GIS Cut Line= 3
      1596342.39      6796295.57      1597092.38      6796501.30
      1598031.21      6796721.05
#Sta/Elev= 30
  4224.1 1945.98  4286.9 1944.48  4299.4 1939.86  4320.1 1935.56  4331.7 1931.05
  4372.0 1923.83  4405.8 1918.71  4434.2 1920.57  4474.7 1917.29  4506.8 1907.55
  4527.5 1906.23  4554.0 1907.73  4588.5 1906.99  4624.5 1904.93  4707.4 1903.03
  4855.6 1903.60  4890.1 1900.30  4895.2 1898.02  4963.0 1898.50  4990.8 1895.93
  4991.3 1895.43  4997.4 1895.93  5035.3 1902.73  5149.0 1902.81  5240.7 1904.74
  5351.0 1904.50  5456.4 1903.85  5654.0 1907.81  5799.7 1911.51  5966.0 1918.58
#Mann=7,-1,0
  4224.1    0.05       0  4624.5    0.12       0  4990.8    0.07       0
  4997.4    0.12       0  5149.0    0.05       0  5351.0    0.12       0
  5654.0    0.05       0
Bank Sta=4990.8,4997.4
Exp/Cntr=0.3,0.1

Type RM Length L Ch R = 1,25714,635,635,635
BEGIN DESCRIPTION:
Elm 01 78 25714.35
END DESCRIPTION:
XS GIS Cut Line= 3
      1596225.11      6796492.54      1596999.39      6796794.61
      1597800.71      6797115.49
#Sta/Elev= 30
  4172.5 1917.86  4200.3 1918.75  4254.6 1918.39  4290.5 1915.41  4309.0 1916.11
  4314.3 1913.69  4333.4 1912.11  4344.2 1907.90  4368.7 1905.19  4406.1 1903.25
  4531.7 1901.01  4687.6 1900.59  4730.6 1899.10  4857.8 1900.96  4870.1 1899.76
  4887.7 1896.12  4902.3 1896.36  4917.5 1894.59  4942.0 1895.40  4998.1 1893.45
  4998.6 1892.95  5004.8 1893.45  5009.7 1893.88  5020.9 1897.94  5026.0 1901.06
  5246.7 1900.49  5311.3 1901.25  5569.8 1907.58  5828.1 1917.22  5866.8 1919.61
#Mann=5,-1,0
  4172.5    0.05       0  4406.1    0.12       0  4998.1    0.07       0
  5004.8    0.12       0  5020.9    0.05       0
Bank Sta=4998.1,5004.8
Exp/Cntr=0.3,0.1

Type RM Length L Ch R = 1,25079,763,763,763
BEGIN DESCRIPTION:
Elm 01 78 25078.93
END DESCRIPTION:
XS GIS Cut Line= 4
      1596166.74      6796496.26      1596510.49      6797298.34
      1596784.72      6797358.11      1597553.45      6797901.85
#Sta/Elev= 30
  3846.7 1913.37  3946.5 1911.15  3977.8 1906.91  4083.0 1902.43  4470.8 1897.52
  4592.5 1896.74  4631.9 1901.79  4740.3 1903.29  4745.4 1901.07  4775.1 1903.91
  4795.6 1901.05  4833.3 1902.55  4838.4 1899.11  4857.0 1900.22  4882.3 1897.15
  4975.4 1897.47  4980.5 1894.13  5003.2 1890.82  5004.0 1888.65  5004.5 1888.15
  5010.9 1888.65  5022.3 1893.56  5043.2 1897.16  5064.1 1892.83  5108.4 1896.67
  5142.3 1896.28  5358.2 1908.10  5444.4 1923.88  5646.3 1926.01  5941.6 1921.57
#Mann=5,-1,0
  3846.7    0.05       0  4470.8    0.12       0  5004.0    0.07       0
  5010.9    0.12       0  5142.3    0.05       0
Bank Sta=5004,5010.9
Exp/Cntr=0.3,0.1

Type RM Length L Ch R = 1,24316,632,632,632
BEGIN DESCRIPTION:
Elm 01 78 24316.45
END DESCRIPTION:
XS GIS Cut Line= 3
      1595466.21      6797121.25      1596161.54      6797647.30
      1597247.44      6798030.10
#Sta/Elev= 30
  4135.2 1918.76  4232.6 1915.54  4288.8 1910.04  4346.8 1913.04  4403.3 1909.96
  4409.6 1906.63  4417.8 1906.61  4424.1 1903.21  4438.7 1900.78  4447.0 1901.78
  4488.6 1895.88  4532.3 1893.03  4660.3 1892.12  4682.1 1894.43  4883.0 1889.87
  4923.7 1891.38  5016.7 1885.77  5017.2 1885.27  5023.7 1885.77  5046.4 1888.48
  5082.0 1891.89  5118.3 1890.39  5180.4 1893.17  5254.6 1892.08  5307.7 1894.51
  5519.4 1895.60  5636.4 1902.42  5784.8 1904.02  5894.5 1909.46  6158.5 1919.31
#Mann=7,-1,0
  4135.2    0.05       0  4883.0    0.12       0  5016.7    0.07       0
  5023.7    0.12       0  5046.4    0.05       0  5519.4    0.12       0
  5894.5    0.05       0
Bank Sta=5016.7,5023.7
Exp/Cntr=0.3,0.1

Type RM Length L Ch R = 1,23684,487,487,487
BEGIN DESCRIPTION:
Elm 01 78 23684.18
END DESCRIPTION:
XS GIS Cut Line= 3
      1594875.51      6797413.21      1595625.51      6797923.63
      1596878.09      6798025.19
#Sta/Elev= 30
  4097.3 1921.37  4114.8 1916.58  4135.7 1913.54  4186.6 1911.33  4201.5 1907.64
  4237.5 1907.09  4279.4 1903.16  4360.1 1906.14  4459.6 1899.10  4503.8 1901.02
  4611.6 1899.25  4662.4 1897.22  4683.4 1894.17  4719.3 1894.27  4785.1 1891.42
  4834.5 1886.05  4863.0 1887.83  4987.9 1884.22  4988.4 1883.72  4995.7 1884.22
  5004.0 1885.64  5060.2 1886.95  5091.3 1886.89  5124.9 1888.25  5264.9 1888.32
  5545.8 1891.55  5766.5 1891.56  6068.3 1899.43  6117.6 1901.88  6261.2 1905.05
#Mann=6,-1,0
  4097.3    0.05       0  4987.9    0.05       0  4995.7    0.05       0
  5060.2    0.12       0  5091.3    0.05       0  6068.3    0.12       0
Bank Sta=4987.9,4995.7
Exp/Cntr=0.3,0.1

Type RM Length L Ch R = 1,23197,509,509,509
BEGIN DESCRIPTION:
Elm 01 78 23196.99
END DESCRIPTION:
XS GIS Cut Line= 3
      1594393.72      6797910.60      1595406.76      6798243.94
      1596719.28      6798415.82
#Sta/Elev= 30
  3936.4 1913.18  4102.5 1901.80  4330.3 1892.65  4356.8 1889.32  4362.0 1890.53
  4379.9 1888.42  4401.0 1888.09  4420.4 1890.21  4483.9 1889.69  4711.7 1886.25
  4775.3 1883.27  4838.9 1884.67  4875.9 1883.52  4948.4 1884.31  4971.3 1883.46
  4997.5 1880.34  4998.0 1879.84  5005.3 1880.34  5021.3 1883.22  5148.5 1885.98
  5192.7 1884.54  5263.3 1886.15  5616.5 1886.17  5843.0 1888.45  5916.8 1891.63
  6090.3 1894.88  6110.5 1897.10  6153.4 1897.21  6326.2 1906.59  6326.6 1906.59
#Mann=4,-1,0
  3936.4    0.05       0  4997.5    0.05       0  5005.3    0.05       0
  6326.2    0.12       0
Bank Sta=4997.5,5005.3
Exp/Cntr=0.3,0.1

Type RM Length L Ch R = 1,22688,552,552,552
BEGIN DESCRIPTION:
Elm 01 78 22687.68
END DESCRIPTION:
XS GIS Cut Line= 3
      1594148.93      6798353.31      1595086.45      6798608.53
      1596674.95      6798764.77
#Sta/Elev= 30
  4029.4 1929.03  4063.9 1930.60  4201.5 1930.57  4217.8 1927.73  4243.0 1926.65
  4257.6 1923.98  4292.2 1912.65  4331.9 1904.76  4377.7 1898.55  4446.0 1891.99
  4543.5 1886.22  4616.1 1883.60  4748.6 1882.02  4854.4 1878.01  4942.2 1880.35
  5009.6 1880.23  5015.7 1877.20  5016.2 1876.70  5023.6 1877.20  5045.8 1880.39
  5080.0 1879.73  5147.1 1882.08  5349.7 1882.89  5572.3 1881.18  6064.0 1885.43
  6235.5 1891.94  6396.3 1894.80  6416.4 1896.72  6479.3 1897.97  6597.2 1903.50
#Mann=3,-1,0
  4029.4    0.05       0  5015.7    0.03       0  5023.6    0.05       0
Bank Sta=5015.7,5023.6
Exp/Cntr=0.3,0.1

Type RM Length L Ch R = 1,22136,430,430,430
BEGIN DESCRIPTION:
Elm 01 78 22136.08
END DESCRIPTION:
XS GIS Cut Line= 3
      1594079.51      6798632.62      1594707.11      6798939.91
      1596519.60      6798968.55
#Sta/Elev= 30
  4304.3 1907.27  4321.5 1903.67  4327.5 1904.62  4355.6 1902.59  4440.0 1915.05
  4462.5 1915.92  4558.1 1899.09  4580.6 1896.60  4597.6 1898.49  4603.1 1896.43
  4620.1 1896.67  4732.6 1880.71  4783.2 1880.55  4878.8 1876.81  4968.8 1877.83
  4981.7 1874.55  4982.2 1874.05  4989.7 1874.55  4999.1 1876.94  5021.0 1877.73
  5541.0 1881.05  5621.1 1878.82  5781.1 1879.40  5851.1 1878.14  5911.6 1879.36
  6078.5 1880.69  6201.1 1882.06  6351.1 1886.10  6511.2 1887.41  6815.8 1894.87
#Mann=5,-1,0
  4304.3    0.05       0  4981.7    0.05       0  4989.7    0.05       0
  5911.6    0.12       0  6078.5    0.05       0
Bank Sta=4981.7,4989.7
Exp/Cntr=0.3,0.1

Type RM Length L Ch R = 1,21706,393,393,393
BEGIN DESCRIPTION:
Elm 01 78 21705.73
END DESCRIPTION:
XS GIS Cut Line= 3
      1593923.23      6799244.59      1594655.03      6799252.41
      1596537.87      6799208.13
#Sta/Elev= 30
  4268.8 1919.13  4310.6 1920.69  4330.6 1918.89  4390.6 1901.76  4440.6 1891.18
  4480.6 1886.05  4520.6 1882.84  4770.6 1874.35  4820.6 1875.85  4870.6 1874.91
  4890.6 1876.33  4900.6 1875.42  4960.6 1876.20  4986.6 1872.42  4987.1 1871.92
  4994.6 1872.42  4998.1 1874.46  5003.1 1874.46  5010.6 1876.68  5110.6 1877.51
  5510.8 1877.34  5650.8 1876.28  5710.8 1876.67  5740.8 1878.07  5930.9 1878.70
  6060.9 1880.93  6391.0 1883.77  6491.0 1886.03  6621.1 1887.00  6884.0 1894.63
#Mann=3,-1,0
  4268.8    0.05       0  4986.6    0.05       0  4994.6    0.05       0
Bank Sta=4986.6,4994.6
Exp/Cntr=0.3,0.1

Type RM Length L Ch R = 1,21313,833,833,833
BEGIN DESCRIPTION:
Elm 01 78 21313.38
END DESCRIPTION:
XS GIS Cut Line= 3
      1593790.44      6799450.32      1594350.34      6799442.51
      1596548.23      6799416.47
#Sta/Elev= 30
  4440.6 1917.60  4495.2 1918.79  4555.2 1917.59  4675.2 1881.21  4715.2 1875.72
  4825.2 1873.11  4875.2 1874.17  4915.2 1873.05  4958.8 1867.08  4959.3 1866.58
  4966.8 1867.08  4985.2 1867.33  5000.4 1871.94  5025.2 1874.14  5065.2 1875.17
  5435.2 1875.35  5645.3 1877.61  5675.3 1877.22  5705.3 1869.57  5735.3 1869.50
  5755.3 1870.86  5785.3 1876.98  5825.3 1874.93  5845.3 1876.44  5905.3 1875.50
  5935.3 1877.23  6105.3 1877.06  6795.3 1883.33  7005.4 1887.33  7198.6 1894.41
#Mann=3,-1,0
  4440.6    0.05       0  4958.8    0.03       0  4966.8    0.05       0
Bank Sta=4958.8,4966.8
Exp/Cntr=0.3,0.1

Type RM Length L Ch R = 1,20480,460,460,460
BEGIN DESCRIPTION:
Elm 01 78 20480.48
END DESCRIPTION:
XS GIS Cut Line= 3
      1593475.62      6799611.97      1594159.63      6800080.70
      1595110.49      6800386.09
#Sta/Elev= 30
  4168.2 1879.91  4381.0 1875.40  4524.4 1870.27  4963.8 1869.51  4969.8 1868.34
  4974.6 1863.71  4975.1 1863.21  4982.7 1863.71  4984.8 1864.94  5001.4 1864.16
  5055.6 1866.06  5076.6 1869.47  5135.0 1870.54  5286.6 1870.00  5327.7 1869.09
  5339.1 1867.13  5370.7 1865.73  5402.4 1865.35  5429.2 1865.96  5486.2 1864.86
  5601.7 1868.77  5691.3 1865.64  5696.6 1866.83  5723.4 1864.94  5787.7 1865.79
  5825.0 1867.89  5857.1 1871.87  5884.0 1879.16  5906.3 1882.33  5996.1 1885.03
#Mann=3,-1,0
  4168.2    0.05       0  4974.6    0.05       0  4982.7    0.05       0
Bank Sta=4974.6,4982.7
Exp/Cntr=0.3,0.1

Type RM Length L Ch R = 1,20020,609,609,609
BEGIN DESCRIPTION:
Elm 01 78 20019.89
END DESCRIPTION:
XS GIS Cut Line= 3
      1593076.33      6799934.89      1593833.24      6800361.95
      1595010.17      6800490.41
#Sta/Elev= 30
  4131.9 1886.11  4228.9 1881.50  4288.1 1875.13  4315.5 1875.66  4374.7 1871.82
  4405.9 1872.48  4486.3 1868.51  4676.6 1866.80  4727.4 1862.67  4735.9 1865.89
  4741.6 1865.08  4763.3 1867.60  4897.6 1866.63  4919.3 1865.03  4934.1 1866.95
  4974.5 1861.65  4975.0 1861.15  4982.6 1861.65  5032.9 1867.05  5173.8 1869.83
  5354.8 1868.22  5505.7 1863.62  5626.4 1866.87  5717.0 1865.02  5737.1 1862.59
  5777.3 1864.12  6024.1 1865.35  6059.0 1869.95  6089.2 1880.84  6184.9 1882.42
#Mann=3,-1,0
  4131.9    0.05       0  4974.5    0.05       0  4982.6    0.05       0
Bank Sta=4974.5,4982.6
Exp/Cntr=0.3,0.1

Type RM Length L Ch R = 1,19411,485,485,485
BEGIN DESCRIPTION:
Elm 01 78 19411.37
END DESCRIPTION:
XS GIS Cut Line= 3
      1592111.06      6800337.66      1593361.02      6800691.82
      1594708.28      6800643.20
#Sta/Elev= 30
  3703.7 1870.56  3835.5 1871.75  3942.5 1869.14  4071.6 1868.08  4102.8 1869.46
  4122.6 1867.72  4127.8 1869.07  4133.9 1867.36  4161.7 1868.91  4234.8 1868.66
  4248.3 1867.26  4273.9 1868.95  4425.2 1866.53  4965.4 1865.55  5021.9 1858.67
  5022.4 1858.17  5031.9 1858.67  5066.9 1864.04  5076.9 1863.02  5116.9 1864.84
  5197.0 1863.07  5244.7 1864.83  5537.2 1865.84  5787.4 1864.92  5917.4 1862.49
  6107.6 1864.28  6167.6 1861.51  6217.6 1863.99  6297.7 1877.55  6351.0 1878.47
#Mann=3,-1,0
  3703.7    0.05       0  5021.9    0.03       0  5031.9    0.05       0
Bank Sta=5021.9,5031.9
Exp/Cntr=0.3,0.1

Type RM Length L Ch R = 1,18926,514,514,514
BEGIN DESCRIPTION:
Elm 01 78 18926.23
END DESCRIPTION:
XS GIS Cut Line= 3
      1592549.69      6801079.49      1593205.98      6801123.76
      1593885.70      6800938.86
#Sta/Elev= 30
  4344.7 1864.90  4401.0 1864.99  4440.2 1863.18  4530.4 1862.35  4570.5 1861.05
  4821.1 1861.75  4831.1 1859.90  4844.4 1855.86  4846.1 1854.43  4846.6 1853.93
  4856.2 1854.43  4871.2 1854.59  4881.2 1855.88  4911.3 1862.00  4921.3 1863.25
  4951.4 1861.45  4971.4 1857.79  4988.8 1856.99  4999.5 1858.11  5006.0 1857.13
  5022.2 1859.83  5040.6 1861.71  5177.6 1862.40  5250.2 1864.58  5268.9 1862.54
  5274.1 1863.36  5348.4 1863.09  5428.0 1861.00  5602.5 1864.45  5706.9 1865.29
#Mann=3,-1,0
  4344.7    0.05       0  4846.1    0.03       0  4856.2    0.05       0
Bank Sta=4846.1,4856.2
Exp/Cntr=0.3,0.1

Type RM Length L Ch R = 1,18412,341,341,341
BEGIN DESCRIPTION:
Elm 01 78 18412.14
END DESCRIPTION:
XS GIS Cut Line= 3
      1592062.70      6801445.80      1592953.38      6801557.79
      1593726.85      6801328.61
#Sta/Elev= 30
  4099.2 1865.11  4232.3 1864.97  4323.2 1864.19  4353.5 1863.18  4363.6 1864.38
  4373.6 1864.31  4393.1 1862.91  4414.0 1863.14  4494.6 1862.21  4634.3 1860.00
  4639.3 1860.60  4686.1 1858.88  4756.6 1857.99  4800.1 1858.18  4817.1 1858.85
  4827.2 1858.26  4897.7 1858.76  4955.8 1858.17  4960.9 1858.60  5003.5 1854.82
  5004.0 1854.32  5013.6 1854.32  5014.1 1854.82  5040.3 1858.42  5052.4 1859.07
  5426.2 1859.46  5572.0 1860.35  5643.7 1861.76  5707.8 1861.38  5803.6 1862.20
#Mann=3,-1,0
  4099.2    0.05       0  5003.5    0.03       0  5014.1    0.05       0
Bank Sta=5003.5,5014.1
Exp/Cntr=0.3,0.1
