--- Elm 01 91.prj (project) ---

Proj Title=Elm 01 91 Base Level Engineering
Current Plan=p01
Default Exp/Contr=0.3,0.1
English Units
Geom File=g01
Flow File=f01
Plan File=p01
Y Axis Title=Elevation
X Axis Title(PF)=Main Channel Distance
X Axis Title(XS)=Station
BEGIN DESCRIPTION:
Elm 01 91
END DESCRIPTION:
DSS Export Rating Curves= 0
DSS Export Rating Curve Sorted= 0
DSS Export Volume Flow Curves= 0
DXF OffsetX= 0
DXF OffsetY= 0
DXF ScaleX= 1
DXF ScaleY= 10

--- Elm 01 91.p01 (plan) ---

Plan Title=Multiple Run
Short Identifier=Multiple
Geom File=g01
Flow File=f01
Subcritical Flow
K Sum by GR= 0
Std Step Tol= 0.01
Critical Tol= 0.01
Num of Std Step Trials= 20
Max Error Tol= 0.3
Flow Tol Ratio= 0.001
Split Flow NTrial= 30
Split Flow Tol= 0.02
Split Flow Ratio= 0.02
Log Output Level= 0
Friction Slope Method= 1
Unsteady Friction Slope Method= 2
Unsteady Bridges Friction Slope Method= 1
Parabolic Critical Depth
Global Vel Dist=  1 , 1 , 1
Global Log Level= 0
CheckData=True
Encroach Param= -1, 0, 0, 0
BEGIN DESCRIPTION:
Multiple Run
END DESCRIPTION:

--- Elm 01 91.f01 (steady flow) ---

Flow Title=Multiple
Program Version=4.10
Number of Profiles= 7
Profile Names=10-year,25-year,50-year,1pct_min,100-year,1pct_plu,500-year
River Rch & RM=Elm 01 91,Reach-1         ,46795
     412     602     768     609     977    1340    1600
River Rch & RM=Elm 01 91,Reach-1         ,46047
     486     709     904     715    1150    1580    1870
River Rch & RM=Elm 01 91,Reach-1         ,40371
     543     799    1020     812    1300    1790    2140
River Rch & RM=Elm 01 91,Reach-1         ,38836
     661     977    1260     999    1600    2200    2640
River Rch & RM=Elm 01 91,Reach-1         ,38069
     661     977    1260     999    1600    2200    2640
River Rch & RM=Elm 01 91,Reach-1         ,31953
     735    1090    1400    1110    1780    2450    2940
River Rch & RM=Elm 01 91,Reach-1         ,28489
     776    1150    1480    1170    1880    2590    3090
River Rch & RM=Elm 01 91,Reach-1         ,27231
     776    1150    1480    1170    1880    2590    3090
River Rch & RM=Elm 01 91,Reach-1         ,22961
    1070    1590    2050    1630    2620    3600    4320
River Rch & RM=Elm 01 91,Reach-1         ,13534
    1060    1570    2020    1600    2570    3530    4220
River Rch & RM=Elm 01 91,Reach-1         ,11574
    1160    1720    2210    1750    2810    3870    4610
River Rch & RM=Elm 01 91,Reach-1         ,22
    2080    3140    4080    3270    5240    7210    8770
Boundary for River Rch & Prof#=Elm 01 91,Reach-1         , 1
Up Type= 0
Dn Type= 3
Dn Slope=0.001
Boundary for River Rch & Prof#=Elm 01 91,Reach-1         , 2
Up Type= 0
Dn Type= 3
Dn Slope=0.001
Boundary for River Rch & Prof#=Elm 01 91,Reach-1         , 3
Up Type= 0
Dn Type= 3
Dn Slope=0.001
Boundary for River Rch & Prof#=Elm 01 91,Reach-1         , 4
Up Type= 0
Dn Type= 3
Dn Slope=0.001
Boundary for River Rch & Prof#=Elm 01 91,Reach-1         , 5
Up Type= 0
Dn Type= 3
Dn Slope=0.001
Boundary for River Rch & Prof#=Elm 01 91,Reach-1         , 6
Up Type= 0
Dn Type= 3
Dn Slope=0.001
Boundary for River Rch & Prof#=Elm 01 91,Reach-1         , 7
Up Type= 0
Dn Type= 3
Dn Slope=0.001
DSS Import GetInterval= 0
DSS Import GetPeak= 0
DSS Import FillOption= 0

--- Elm 01 91.g01 (geometry) ---

Geom Title=Existing Conditions
Program Version=4.10

River Reach=Elm 01 91       ,Reach-1
Reach XY= 30
        1602705.        6782788.      1603853.08      6785693.98
        1603658.       6786986.6      1604799.64       6787985.3
      1605504.51      6789853.22      1604904.51      6790558.12
      1605404.14      6791098.31      1605256.95      6792382.11
      1606148.03      6793088.25      1605208.53      6793039.45
      1605347.69      6794788.04      1604712.58      6796041.35
      1606247.33      6797581.48      1606058.03      6798136.61
      1606960.44      6799332.75      1607599.55      6799235.53
      1607407.16      6800432.57      1608197.54      6800931.95
      1608355.53      6801862.86      1607756.67      6803482.33
      1608507.46      6803243.45      1609291.43      6804574.53
      1610652.92      6805193.49       1609710.4      6805985.57
      1609549.78      6807183.45      1609054.73      6807006.45
      1609210.25      6808032.56      1609736.59      6807587.63
      1610299.54      6808085.55        1610305.        6809038.

Type RM Length L Ch R = 1 ,46795   ,156,156,156
BEGIN DESCRIPTION:
Elm 01 91 46699.719
END DESCRIPTION:
XS GIS Cut Line= 3
      1602344.78      6782842.36      1602704.89      6782813.06
      1603054.39      6782801.12
#Sta/Elev= 30
  4638.7 2046.74    4669 2045.57  4709.1 2041.48  4749.2 2039.31  4799.4 2035.24
  4819.5 2034.61  4849.6 2031.78  4869.7 2025.49    4876 2024.86  4881.1  2022.5
  4889.7 2021.09  4949.9 2016.89    4978 2012.76  4978.3 2012.26    4982 2012.76
    5000 2013.75  5003.4 2014.96  5010.1 2015.71  5020.1 2014.86  5050.1 2026.63
  5060.1 2028.72  5100.2 2032.15  5120.2 2033.03  5190.2 2033.95  5200.2 2034.93
  5220.2  2034.5  5260.3 2035.81  5270.3 2035.42  5300.3  2036.7  5349.7 2036.56
#Mann= 3 ,-1 , 0
  4638.7     .12       0    4978     .07       0    4982     .12       0
Bank Sta=4978,4982
XS Rating Curve= 0 ,0
Exp/Cntr=0.3,0.1

Type RM Length L Ch R = 1 ,46639   ,205,205,205
BEGIN DESCRIPTION:
Elm 01 91 46639.47
END DESCRIPTION:
XS GIS Cut Line= 3
      1602423.96      6783032.25      1602726.73      6782961.71
       1603009.9      6782900.96
#Sta/Elev= 30
  4687.9 2050.81  4726.8 2049.36  4731.9 2049.95  4740.3 2049.26  4817.1 2049.51
  4853.3  2047.6  4859.6  2046.4  4864.8  2046.6  4935.4 2020.66  4944.8 2017.63
  4949.9 2017.04  4955.9 2013.69  4964.2 2011.49  4964.5 2010.99    4968 2010.99
  4968.2 2011.49  4986.7 2012.96  4992.5 2012.19  5007.2 2013.59  5027.7  2018.8
  5036.6    2020  5041.7 2021.65  5058.4 2022.79    5086 2025.98  5091.1 2029.06
    5130 2029.44  5211.8 2028.75  5273.2 2031.07  5278.5 2031.78  5288.4 2031.59
#Mann= 3 ,-1 , 0
  4687.9     .12       0  4964.2     .07       0  4968.2     .12       0
Bank Sta=4964.2,4968.2
XS Rating Curve= 0 ,0
Exp/Cntr=0.3,0.1

Type RM Length L Ch R = 1 ,46434   ,208,208,208
BEGIN DESCRIPTION:
Elm 01 91 46433.91
END DESCRIPTION:
XS GIS Cut Line= 3
      1602638.29      6783212.72      1602872.69      6783106.81
      1603088.86      6782999.16
#Sta/Elev= 30
  4741.5 2033.83  4748.9  2033.9  4781.8  2031.9  4803.7 2029.78  4816.9 2029.69
  4834.6 2028.34  4840.1 2028.68  4857.7  2027.1  4863.2 2027.31  4869.6 2025.97
  4891.8 2023.52  4902.5 2023.58  4924.4 2021.58  4955.6 2017.35  4961.1 2015.83
  4968.3 2012.65  4982.2  2008.8  4982.5  2008.3    4986  2008.3  4986.2  2008.8
  5007.1 2010.99  5023.6 2014.43  5029.5 2018.09    5035 2020.65  5051.8  2024.2
    5147 2027.41  5163.8  2027.4  5191.8 2028.88  5230.9 2028.14  5240.2 2028.77
#Mann= 3 ,-1 , 0
  4741.5     .12       0  4982.2     .07       0  4986.2     .12       0
Bank Sta=4982.2,4986.2
XS Rating Curve= 0 ,0
Exp/Cntr=0.3,0.1

Type RM Length L Ch R = 1 ,46226   ,179,179,179
BEGIN DESCRIPTION:
Elm 01 91 46225.71
END DESCRIPTION:
XS GIS Cut Line= 3
      1602752.09       6783376.6      1602918.79      6783300.19
      1603105.61      6783197.41
#Sta/Elev= 30
  4816.6 2025.72  4853.8 2025.38  4871.3 2024.31  4885.8 2024.13  4894.3 2023.25
  4922.8  2023.3  4929.8 2022.66  4940.3  2020.9  4951.8 2020.39  4962.8 2018.66
  4968.8 2015.74  4974.3 2017.63  4984.8 2014.03  4991.8 2010.28  5007.1 2009.36
  5011.8 2007.58  5012.1 2007.08  5015.6 2007.08  5015.8 2007.58  5029.9 2009.11
  5035.6 2010.74  5041.3 2013.61  5051.7  2015.7    5087 2017.19    5101 2019.45
  5109.8 2020.23  5144.5 2021.39  5166.9 2021.05  5204.2 2021.53  5213.2 2020.82
#Mann= 3 ,-1 , 0
  4816.6     .12       0  5011.8     .07       0  5015.8     .12       0
Bank Sta=5011.8,5015.8
XS Rating Curve= 0 ,0
Exp/Cntr=0.3,0.1

Type RM Length L Ch R = 1 ,46047   ,208,208,208
BEGIN DESCRIPTION:
Elm 01 91 46047.28
END DESCRIPTION:
XS GIS Cut Line= 3
      1602896.72      6783491.53      1603061.32      6783397.07
      1603365.48      6783235.27
#Sta/Elev= 30
  4810.6 2021.35  4864.2 2019.57  4877.8 2017.85  4891.6 2018.62  4958.5 2016.89
  4966.3 2015.39  4972.1 2013.23  4987.9 2011.42  4993.7 2008.31  5004.7 2007.86
  5009.6 2006.69  5013.8 2006.56  5014.1 2006.06  5017.9 2006.56  5038.5 2007.86
  5061.2 2007.97  5069.9 2009.28  5075.6 2011.39  5091.9 2015.61  5097.5 2016.07
  5129.1 2015.97  5135.8 2014.45  5151.8 2014.68  5163.4  2015.9  5174.1  2015.9
  5179.8 2016.84  5201.7 2016.27    5218 2015.03  5276.4 2018.97  5344.9 2020.43
#Mann= 3 ,-1 , 0
  4810.6     .12       0  5013.8     .07       0  5017.9     .12       0
Bank Sta=5013.8,5017.9
XS Rating Curve= 0 ,0
Exp/Cntr=0.3,0.1

Type RM Length L Ch R = 1 ,45839   ,250,250,250
BEGIN DESCRIPTION:
Elm 01 91 45838.81
END DESCRIPTION:
XS GIS Cut Line= 3
      1602887.93      6783732.01      1603209.98      6783542.77
      1603434.31      6783371.94
#Sta/Elev= 30
  4626.3  2027.6  4634.5 2027.54  4669.5 2024.44  4700.8 2022.58  4706.6 2021.36
  4728.1 2019.22  4786.7 2017.56  4854.9 2013.99  4866.7 2012.12  4876.6  2011.4
  4882.4 2009.13  4889.7 2009.94  4903.9  2008.2  4919.5 2007.46  4993.8 2006.67
  5014.2 2005.67  5020.5 2006.27    5033 2005.58  5033.2 2005.08  5036.8 2005.08
  5037.1 2005.58  5056.4 2006.39  5070.4 2008.23  5078.6 2010.52  5084.9 2011.01
  5093.2 2013.04    5114 2014.62    5157 2015.43  5257.4 2015.08  5281.8 2015.76
#Mann= 3 ,-1 , 0
  4626.3     .12       0    5033     .07       0  5037.1     .12       0
Bank Sta=5033,5037.1
XS Rating Curve= 0 ,0
Exp/Cntr=0.3,0.1

Type RM Length L Ch R = 1 ,45589   ,302,302,302
BEGIN DESCRIPTION:
Elm 01 91 45589.47
END DESCRIPTION:
XS GIS Cut Line= 3
      1602985.99      6783901.29      1603303.73      6783756.31
      1603517.26      6783559.27
#Sta/Elev= 30
  4649.2 2030.86  4659.1 2033.07  4666.9 2036.09  4672.4 2036.32  4681.1  2034.6
  4703.1 2025.88    4713 2023.07    4747  2015.6  4762.4 2013.84    4770 2014.36
    4802 2013.35  4900.9 2006.71  4954.3 2007.19  4977.4 2005.35  5024.6 2003.76
  5024.9 2003.26  5028.8 2003.76  5061.9 2004.28  5068.7 2005.42    5076 2004.75
  5082.8 2006.03  5104.4 2005.29  5139.5 2007.75  5146.9  2007.4  5153.7 2008.74
  5161.1 2008.41  5167.9 2009.62  5189.5 2009.57  5267.1 2012.66    5289 2012.62
#Mann= 4 ,-1 , 0
  4649.2     .05       0  4762.4     .12       0  5024.6     .07       0
  5028.8     .12       0
Bank Sta=5024.6,5028.8
XS Rating Curve= 0 ,0
Exp/Cntr=0.3,0.1

Type RM Length L Ch R = 1 ,45287   ,314,314,314
BEGIN DESCRIPTION:
Elm 01 91 45286.61
END DESCRIPTION:
XS GIS Cut Line= 3
      1602950.95      6784042.94      1603204.39      6784021.42
      1603759.29      6783899.88
#Sta/Elev= 30
  4745.4 2037.64  4819.7 2031.52  4858.9 2022.68  4863.9 2023.02  4869.9 2020.45
  4922.6 2011.31  4940.1 2008.97  4978.2 2000.84  4983.2 2001.83  4990.3 1999.75
  5010.6 2000.41    5029 1999.23  5029.3 1998.73  5033.2 1999.23  5081.5 2002.62
  5135.6 2004.52  5174.3 2003.69  5179.4 2004.46  5205.1 2000.49    5287 2003.11
    5328 2001.85  5358.7 2003.74    5365 2005.88  5370.1 2005.17  5389.4 2009.18
  5430.3 2011.27  5491.8 2011.88  5512.2 2013.05  5532.7 2016.06  5567.8 2016.26
#Mann= 4 ,-1 , 0
  4745.4     .05       0  4922.6     .12       0    5029     .07       0
  5033.2     .12       0
Bank Sta=5029,5033.2
XS Rating Curve= 0 ,0
Exp/Cntr=0.3,0.1

Type RM Length L Ch R = 1 ,44973   ,231,231,231
BEGIN DESCRIPTION:
Elm 01 91 44973.11
END DESCRIPTION:
XS GIS Cut Line= 3
      1602885.31       6784282.6      1603384.44      6784219.23
      1604015.55      6784076.86
#Sta/Elev= 30
  4496.3  2026.3  4546.4 2025.47    4572 2023.04  4577.1  2023.5  4596.8  2020.9
  4637.1  2017.9  4667.4 2017.85    4748 2010.59  4768.2 2010.27  4798.4 2008.22
  4892.1 2004.52  4939.5 2001.15  4989.9  1998.7  4994.7 1997.08  4995.1 1996.58
  4999.7 1997.08  5020.5  1998.9  5061.5 1997.28    5075 1998.44  5112.8 1997.94
  5118.3 1999.58  5123.4 1999.57  5143.5 2002.03  5215.3  2005.2  5349.8 2009.66
  5369.1 2009.71  5484.6  2014.4  5527.8 2015.31  5543.3 2016.79  5646.4 2022.74
#Mann= 3 ,-1 , 0
  4496.3     .12       0  4994.7     .07       0  4999.7     .12       0
Bank Sta=4994.7,4999.7
XS Rating Curve= 0 ,0
Exp/Cntr=0.3,0.1

Type RM Length L Ch R = 1 ,44742   ,243,243,243
BEGIN DESCRIPTION:
Elm 01 91 44742
END DESCRIPTION:
XS GIS Cut Line= 3
      1602860.83       6784421.3      1603504.26      6784408.28
      1604168.32      6784274.81
#Sta/Elev= 30
  4356.2  2019.1  4400.4  2017.4  4440.4 2017.13  4470.4 2015.09  4480.4 2015.36
  4540.4 2011.19  4590.4 2009.65  4600.4 2008.55  4670.4 2005.16  4700.4 2002.56
  4720.4 2002.13  4765.9 1998.76  4770.9 1999.28  4810.5 1997.12  4960.5 1997.53
  4970.5 1996.51  5002.7 1997.17  5038.8 1996.23  5039.2 1995.73  5043.8 1996.23
  5071.9 2000.47  5092.3 2001.76  5173.8 2004.26  5306.5 2006.06  5316.7 2006.95
  5347.3  2007.6  5377.3 2007.13  5382.4 2008.47  5469.7  2011.8  5677.1 2023.65
#Mann= 3 ,-1 , 0
  4356.2     .12       0  5038.8     .07       0  5043.8     .12       0
Bank Sta=5038.8,5043.8
XS Rating Curve= 0 ,0
Exp/Cntr=0.3,0.1

Type RM Length L Ch R = 1 ,44499   ,317,317,317
BEGIN DESCRIPTION:
Elm 01 91 44498.69
END DESCRIPTION:
XS GIS Cut Line= 3
      1602961.72      6784553.68      1603404.43      6784614.44
       1604165.1      6784473.38
#Sta/Elev= 30
  4552.5 2012.81  4596.2 2009.99  4621.2 2009.57  4636.6  2007.6  4666.8 2006.34
  4676.9 2005.02  4717.3 2003.75  4757.7 1997.93  4765.4 1998.61  4770.5 2000.23
  4777.9 1999.26  4888.9 1995.87  4979.7 1994.64  4986.8 1991.53  4991.8 1993.53
  4997.1 1991.54  5008.7 1991.43  5009.1 1990.93  5013.7 1991.43  5030.4 1994.55
  5091.5 1995.24  5128.2 1996.76  5256.7 2000.52  5528.8 2004.55  5612.9 2008.57
  5620.3 2009.68  5665.7 2010.19  5681.4 2012.14  5752.6 2014.59    5773 2016.37
#Mann= 5 ,-1 , 0
  4552.5     .12       0  5008.7     .07       0  5013.7     .12       0
  5128.2     .05       0  5256.7     .12       0
Bank Sta=5008.7,5013.7
XS Rating Curve= 0 ,0
Exp/Cntr=0.3,0.1

Type RM Length L Ch R = 1 ,44182   ,218,218,218
BEGIN DESCRIPTION:
Elm 01 91 44182.27
END DESCRIPTION:
XS GIS Cut Line= 3
      1602860.99      6784822.34      1603604.52      6784852.29
      1604350.27      6784706.52
#Sta/Elev= 30
  4255.6 2007.29  4279.6 2007.56  4319.7  2005.2  4359.7 2005.27  4379.7 2003.69
  4409.7 2002.74  4449.8 2003.59  4489.8 2000.96  4522.7 2001.73  4549.9 1999.25
  4579.9 2000.08  4599.9 1998.06  4629.9 1996.68    4690 1996.56  4796.7 1993.42
  4840.1 1991.05  5028.3 1989.42  5028.6 1988.92  5033.3 1989.42    5081 1994.55
  5112.3 1997.87  5234.6 1998.06  5313.5 1999.26  5397.6 2001.18  5448.6 2001.41
    5581 2005.53  5652.3 2009.36  5727.3  2014.8  5754.2 2018.29  5759.6  2020.7
#Mann= 6 ,-1 , 0
  4255.6     .05       0  4796.7     .12       0  5028.3     .07       0
  5033.3     .12       0    5081     .05       0  5313.5     .12       0
Bank Sta=5028.3,5033.3
XS Rating Curve= 0 ,0
Exp/Cntr=0.3,0.1

Type RM Length L Ch R = 1 ,43964   ,249,249,249
BEGIN DESCRIPTION:
Elm 01 91 43964.41
END DESCRIPTION:
XS GIS Cut Line= 3
      1602780.35      6785007.24      1603504.26      6785033.28
      1604440.21      6784830.21
#Sta/Elev= 30
  4275.6 2008.29  4320.3 2005.15  4330.3 2005.52  4350.3 2003.27  4370.3 2003.48
  4400.3 2001.07  4430.3 2001.03  4460.4 1999.15  4490.4 2000.11  4520.4 1998.22
  4573.1 1997.26  4846.3 1992.54  4970.7 1988.63  4978.2 1986.79  4978.6 1986.29
  4983.3 1986.79  4997.8 1987.91  5072.4 1987.92  5154.2 1992.96  5239.2 1995.88
  5420.3 1997.21  5491.9 1998.66  5573.8 2002.07  5686.3 2004.31  5788.7 2010.25
  5829.6 2014.56  5852.7 2018.21  5870.5 2018.23  5907.8 2022.37  5957.7 2024.11
#Mann= 6 ,-1 , 0
  4275.6     .12       0  4573.1     .05       0  4846.3     .12       0
  4978.2     .07       0  4983.3     .12       0  5907.8     .05       0
Bank Sta=4978.2,4983.3
XS Rating Curve= 0 ,0
Exp/Cntr=0.3,0.1

Type RM Length L Ch R = 1 ,43715   ,178,178,178
BEGIN DESCRIPTION:
Elm 01 91 43715.19
END DESCRIPTION:
XS GIS Cut Line= 3
       1602664.2      6785244.65      1603452.41      6785267.22
      1604315.27      6785142.22
#Sta/Elev= 30
  4209.3 2008.49  4220.1 2009.37  4230.1 2007.57  4280.1 2005.91  4300.1 2003.53
  4330.1 2002.94  4350.2 2000.57  4370.2 2001.46  4390.2 1999.01  4470.2 1999.41
  4530.2 1994.71  4601.6 1993.29  4783.5  1990.9  4852.9 1990.21  4900.4 1986.17
  4990.4 1986.22  5028.9 1985.17  5029.3 1984.67  5034.1 1985.17  5081.3 1987.31
  5135.1 1987.42  5161.9 1987.66  5172.2 1988.69    5336  1989.3  5372.6 1989.08
  5377.7 1990.15  5404.6 1988.22  5434.9  1990.6  5583.3 1996.43  5869.7 2004.21
#Mann= 7 ,-1 , 0
  4209.3     .12       0  4601.6     .05       0  4783.5     .12       0
  5028.9     .07       0  5034.1     .12       0  5135.1     .05       0
    5336     .12       0
Bank Sta=5028.9,5034.1
XS Rating Curve= 0 ,0
Exp/Cntr=0.3,0.1

Type RM Length L Ch R = 1 ,43537   ,363,363,363
BEGIN DESCRIPTION:
Elm 01 91 43536.51
END DESCRIPTION:
XS GIS Cut Line= 3
      1602433.35       6785487.7      1603537.48      6785414.79
      1604334.32      6785348.82
#Sta/Elev= 30
  3897.4 2009.89  3939.1 2007.62  3959.2 2008.56  3966.5 2006.31  3971.5 2008.19
  3989.2 2005.39  4099.5 2001.26  4159.6 2001.24  4199.7  1996.8  4229.8 1995.72
  4575.7 1989.02  4740.9  1988.4  4770.9 1989.42  4828.5 1985.95  4921.3 1984.34
  4941.3 1983.21  4958.8 1979.79  4959.2 1979.29    4964 1979.79  4981.4 1983.39
  5061.7 1981.38  5121.9 1981.26    5152 1982.97  5182.1 1981.37  5212.2 1981.89
  5322.5  1985.4  5362.7  1988.6    5443 1991.87  5766.9 2000.79  5803.5 2001.63
#Mann= 5 ,-1 , 0
  3897.4     .05       0  4828.5     .12       0  4958.8     .07       0
    4964     .12       0  5766.9     .05       0
Bank Sta=4958.8,4964
XS Rating Curve= 0 ,0
Exp/Cntr=0.3,0.1

Type RM Length L Ch R = 1 ,43174   ,252,252,252
BEGIN DESCRIPTION:
Elm 01 91 43174.33
END DESCRIPTION:
XS GIS Cut Line= 3
      1602981.89      6785683.89      1603796.16      6785630.07
       1604331.3      6785597.16
#Sta/Elev= 30
  4182.3 1985.83    4495  1985.2  4536.2  1985.7  4696.5 1984.04  4726.6    1984
  4739.2 1984.87  4756.7 1984.47  4786.7 1982.37  4866.9 1980.43    4907 1979.88
    4958 1980.56  4977.1 1979.44  5007.2 1979.42  5014.6 1975.32    5015 1974.82
  5019.4 1974.82  5019.8 1975.32  5037.3 1978.18  5107.4 1979.78  5137.4 1981.95
  5157.5 1984.67  5177.5 1989.53  5207.6 1992.52  5274.6 1997.61  5279.6  1997.1
  5377.9 2001.53    5428 2005.98  5478.1 2007.19  5498.1 2008.78  5534.5 2010.47
#Mann= 4 ,-1 , 0
  4182.3     .05       0  4739.2     .12       0  5014.6     .07       0
  5019.8     .12       0
Bank Sta=5014.6,5019.8
XS Rating Curve= 0 ,0
Exp/Cntr=0.3,0.1

Type RM Length L Ch R = 1 ,42922   ,123,123,123
BEGIN DESCRIPTION:
Elm 01 91 42922.1
END DESCRIPTION:
XS GIS Cut Line= 3
      1603261.65       6785774.6      1603783.75      6785813.66
      1604140.95      6785786.38
#Sta/Elev= 30
    4479 1984.52  4582.6 1984.65  4662.9 1983.72  4743.1 1981.79  4823.3    1982
  4833.3 1980.57    4881 1978.51  4913.6 1976.85  4923.6 1977.43  4953.7 1974.76
  4973.7 1974.97  4996.3 1973.95    5010  1974.4    5015 1973.53  5023.9 1974.55
  5031.2 1973.09  5031.7 1972.59  5036.1 1972.59  5036.5 1973.09    5074 1976.34
  5094.1 1976.51  5134.2 1977.93  5140.9 1980.03  5145.9 1978.32  5164.3 1982.64
  5194.4 1992.32  5244.5 1998.06  5284.6 2003.98  5320.9 2006.91  5360.8 2009.06
#Mann= 5 ,-1 , 0
    4479     .05       0    4881     .12       0  5031.2     .07       0
  5036.5     .12       0  5320.9     .05       0
Bank Sta=5031.2,5036.5
XS Rating Curve= 0 ,0
Exp/Cntr=0.3,0.1

Type RM Length L Ch R = 1 ,42799   ,353,353,353
BEGIN DESCRIPTION:
Elm 01 91 42799.49
END DESCRIPTION:
XS GIS Cut Line= 3
      1603311.08      6785925.64      1603705.62      6785906.11
      1604081.58      6785902.22
#Sta/Elev= 30
  4605.7 1982.92  4619.6 1983.61  4639.7    1983  4679.7    1984  4759.8 1983.83
  4769.8 1983.11  4829.9 1982.56    4920  1978.9    4940 1979.56  4960.1 1979.22
  4980.1 1974.81  5002.9 1973.03  5007.5 1970.58  5007.9 1970.08  5012.8 1970.58
  5020.1 1972.85  5030.1 1974.65  5060.1 1974.04  5080.1 1975.54  5100.1 1975.06
  5140.1 1976.66  5160.1 1976.65  5180.1 1978.21  5210.1 1983.28  5240.1  1986.9
  5270.1 1993.26  5298.2 1997.68  5303.2 1997.13  5340.1 2002.21  5376.7 2004.97
#Mann= 3 ,-1 , 0
  4605.7     .12       0  5007.5     .07       0  5012.8     .12       0
Bank Sta=5007.5,5012.8
XS Rating Curve= 0 ,0
Exp/Cntr=0.3,0.1

Type RM Length L Ch R = 1 ,42446   ,254,254,254
BEGIN DESCRIPTION:
Elm 01 91 42445.91
END DESCRIPTION:
XS GIS Cut Line= 3
      1603462.17      6786074.08      1603947.81      6786137.88
      1604201.55      6786158.59
#Sta/Elev= 30
  4510.3 1981.31  4533.3 1979.05  4553.5 1979.61  4573.7  1979.2  4593.8 1977.77
  4674.5 1975.58  4755.2 1974.48  4765.3 1975.01  4775.4 1973.99  4866.2 1974.91
  4876.2 1974.63  4896.4 1972.07  4946.8  1971.8  4962.3 1970.53  4977.1 1970.88
  4987.2 1968.74  4993.5 1968.16  4993.9 1967.66  4998.8 1968.16  5000.1 1968.16
  5007.3 1972.95  5047.5  1989.1  5057.5 1994.57  5062.8 1999.32  5067.8 1997.96
  5077.6  1999.9  5167.9 2005.76  5189.5 2005.36  5238.1 2006.64  5254.7 2005.83
#Mann= 3 ,-1 , 0
  4510.3     .12       0  4993.5     .07       0  4998.8     .12       0
Bank Sta=4993.5,4998.8
XS Rating Curve= 0 ,0
Exp/Cntr=0.3,0.1

Type RM Length L Ch R = 1 ,42192   ,331,331,331
BEGIN DESCRIPTION:
Elm 01 91 42192.22
END DESCRIPTION:
XS GIS Cut Line= 3
      1603457.55       6786275.9      1603807.83      6786342.31
      1604060.26      6786376.14
#Sta/Elev= 30
  4642.6  1977.1  4683.3 1975.47  4772.3  1970.3  4782.5 1970.29  4787.8 1970.97
  4823.2 1970.61  4840.1  1971.1  4845.2 1970.02  4863.9 1969.74  4897.5 1967.74
  4914.8 1969.32  4955.5 1970.41  4986.1 1969.28  4995.1 1967.31  5000.2 1967.17
  5000.6 1966.67  5005.1 1966.67  5005.5 1967.17  5007.9 1968.01  5036.6 1969.94
  5066.9 1970.89  5075.8 1971.91  5080.8 1972.53  5127.4 1982.83  5147.6 1984.76
  5153.8 1986.07  5158.8  1985.7    5188 1989.68  5231.8 1994.17  5253.8 1997.53
#Mann= 3 ,-1 , 0
  4642.6     .12       0  5000.2     .07       0  5005.5     .12       0
Bank Sta=5000.2,5005.5
XS Rating Curve= 0 ,0
Exp/Cntr=0.3,0.1

Type RM Length L Ch R = 1 ,41861   ,245,245,245
BEGIN DESCRIPTION:
Elm 01 91 41860.61
END DESCRIPTION:
XS GIS Cut Line= 3
      1603332.57      6786510.27      1603609.92      6786489.44
      1604008.37      6786458.19
#Sta/Elev= 30
  4720.7 1976.59  4763.2 1976.33  4773.3 1977.03  4818.1 1976.25  4863.5 1974.46
  4893.6 1972.58  4923.7 1972.01  4943.8 1970.45  4955.1 1968.91  4963.8    1967
  4983.9 1964.26  4991.2 1962.33  4991.6 1961.83  4996.1 1961.83  4996.5 1962.33
  4998.8 1962.33    5014 1966.65    5044 1966.73  5064.1 1968.63  5144.4 1971.88
  5174.4 1972.52  5204.3  1974.1  5209.3  1973.7  5224.6 1974.97  5284.8 1977.96
  5304.8  1980.2  5333.5 1984.96  5338.5 1984.58  5394.3  1990.5  5398.5  1990.5
#Mann= 3 ,-1 , 0
  4720.7     .12       0  4991.2     .07       0  4996.5     .12       0
Bank Sta=4991.2,4996.5
XS Rating Curve= 0 ,0
Exp/Cntr=0.3,0.1

Type RM Length L Ch R = 1 ,41616   ,361,361,361
BEGIN DESCRIPTION:
Elm 01 91 41616.43
END DESCRIPTION:
XS GIS Cut Line= 3
       1603340.1      6786748.77      1603705.73      6786704.29
      1604061.32       6786641.6
#Sta/Elev= 30
    4631 1972.99  4696.4 1973.43  4746.7 1973.13  4761.7 1973.84  4807.2 1973.01
  4843.4 1970.82  4877.7 1970.39  4925.1 1967.72  4930.1 1968.14  4948.2 1966.65
  5001.5 1963.84  5016.2 1960.15  5016.6 1959.65  5021.1 1959.65  5021.5 1960.15
  5039.2 1963.54  5079.8 1966.83  5100.1 1967.03  5118.6 1969.64  5140.7  1973.7
    5161 1975.55  5171.2 1975.49  5201.7 1980.39    5222 1981.99  5237.2  1984.2
  5282.9 1989.03  5291.3 1990.41  5296.4 1990.34  5303.2 1991.67  5360.4  1994.9
#Mann= 3 ,-1 , 0
    4631     .12       0  5016.2     .07       0  5021.5     .12       0
Bank Sta=5016.2,5021.5
XS Rating Curve= 0 ,0
Exp/Cntr=0.3,0.1

Type RM Length L Ch R = 1 ,41255   ,347,347,347
BEGIN DESCRIPTION:
Elm 01 91 41255.18
END DESCRIPTION:
XS GIS Cut Line= 3
        1603446.      6787110.55       1603675.2      6787006.37
      1604136.97      6786708.65
#Sta/Elev= 30
  4749.4 1967.66  4835.4 1968.83    4946 1967.78  4961.7 1964.15    4968 1960.28
  4976.3 1959.56  4976.7 1959.06  4981.6 1959.56  4984.8 1960.88  5036.6 1962.37
  5079.7 1961.31  5152.3 1962.18  5215.7 1965.21  5376.1 1964.99  5391.3  1966.9
  5397.2 1969.43  5412.4 1970.09  5418.4 1973.37  5427.6 1974.17  5433.5 1977.58
  5463.9 1981.65  5469.8 1984.97    5485 1984.06    5491 1986.65  5500.2 1986.56
  5506.1 1988.84  5521.3 1986.76  5527.3 1987.91  5542.4 1985.65  5550.6 1986.98
#Mann= 3 ,-1 , 0
  4749.4     .12       0  4976.3     .07       0  4981.6     .12       0
Bank Sta=4976.3,4981.6
XS Rating Curve= 0 ,0
Exp/Cntr=0.3,0.1

Type RM Length L Ch R = 1 ,40908   ,428,428,428
BEGIN DESCRIPTION:
Elm 01 91 40907.7
END DESCRIPTION:
XS GIS Cut Line= 3
      1603590.08      6787375.41      1603949.44      6787187.92
      1604296.65      6786736.54
#Sta/Elev= 30
  4593.8 1964.08  4618.4 1964.81  4678.3 1964.22  4767.4 1964.77  4877.9 1960.19
  4927.7 1959.42  4944.1 1958.41  4990.8 1958.11  4991.2  1958.1  4991.6  1957.6
  4996.5  1958.1  5060.7 1961.48  5111.9  1961.4  5166.7  1959.6  5174.9 1960.28
  5181.2 1959.42  5195.7 1960.35    5202 1959.12  5216.5 1958.58  5280.9 1959.01
  5338.9  1960.3  5380.6 1964.27  5395.1 1965.13  5409.6  1964.9  5415.9 1966.11
  5420.4 1965.99  5459.4 1969.52  5473.9 1969.38  5523.7 1972.37  5568.6 1972.77
#Mann= 6 ,-1 , 0
  4593.8     .12       0  4990.8     .05       0  4991.2     .05       0
  4996.5     .05       0  5111.9     .12       0  5420.4     .05       0
Bank Sta=4991.2,4996.5
XS Rating Curve= 0 ,0
Exp/Cntr=0.3,0.1

Type RM Length L Ch R = 1 ,40480   ,109,109,109
BEGIN DESCRIPTION:
Elm 01 91 40480.11
END DESCRIPTION:
XS GIS Cut Line= 6
      1603784.35      6787337.45      1604032.99      6787484.18
      1604119.57      6787474.38      1604194.23      6787439.65
      1604444.23      6787151.46      1604730.32      6786636.49
#Sta/Elev= 30
    4542 1963.78  4652.2    1963  4689.3 1961.53  4726.4 1961.33  4732.2 1962.52
  4747.8 1960.85  4753.6 1962.12  4769.3 1960.67  4790.7 1962.24  4821.4 1962.39
  4852.9  1958.2  4888.8 1956.89  4988.4 1952.77  5037.5 1954.93  5098.5 1951.56
  5098.9 1951.06  5103.8 1951.56  5172.3 1953.88  5228.3 1953.13  5278.7 1955.23
  5430.2  1956.3    5452 1957.31  5495.4 1962.11  5538.9 1962.99  5545.8 1962.08
  5560.6 1963.25  5598.4 1962.41    5650 1964.17  5742.5 1966.94  5970.8 1972.98
#Mann= 6 ,-1 , 0
    4542     .12       0  4888.8     .05       0  5098.5     .05       0
  5103.8     .05       0    5650     .12       0  5742.5     .05       0
Bank Sta=5098.5,5103.8
XS Rating Curve= 0 ,0
Exp/Cntr=0.3,0.1

Type RM Length L Ch R = 1 ,40371   ,101,101,101
BEGIN DESCRIPTION:
Elm 01 91 40370.8
END DESCRIPTION:
XS GIS Cut Line= 6
      1603651.55      6787388.24      1604074.44      6787545.56
      1604206.38      6787536.88      1604435.55      6787351.11
      1604560.55      6787165.35      1604713.31      6786828.57
#Sta/Elev= 30
  4320.8 1964.07  4738.1 1960.68  4738.6 1960.18  4743.9 1960.68  4760.6 1965.28
    4766  1962.5  4792.6 1965.78  4842.7 1962.88  4915.9 1965.48  4961.4 1961.69
  5010.9 1965.66    5075 1965.98  5124.3 1962.39  5131.7 1964.36  5138.5 1961.78
  5166.9 1966.03  5242.8 1964.15  5275.2 1961.11  5317.2 1965.11  5332.2 1961.85
  5353.2 1964.91  5368.2 1962.37  5374.2 1964.62  5442.5 1965.15    5448 1961.57
  5471.1 1963.91  5487.3 1961.31  5657.2 1966.24  5665.8  1966.4  5794.1 1968.96
#Mann= 6 ,-1 , 0
  4320.8     .12       0  4738.1     .07       0  4743.9     .12       0
  5242.8     .05       0  5657.2     .12       0  5665.8     .05       0
Bank Sta=4738.1,4743.9
XS Rating Curve= 0 ,0
Exp/Cntr=0.3,0.1

Type RM Length L Ch R = 1 ,40270   ,499,499,499
BEGIN DESCRIPTION:
Elm 01 91 40269.86
END DESCRIPTION:
XS GIS Cut Line= 6
      1603859.18       6787677.5      1604234.16      6787608.06
      1604355.69      6787543.82      1604381.73      6787512.57
      1604638.67      6787168.82      1604817.46      6786896.29
#Sta/Elev= 30
  4442.2    1960  4686.8 1960.81  4739.7 1958.16  4804.2 1957.24  4889.9    1955
  4936.7 1952.83  4964.9 1953.76  5004.8 1951.28  5005.3 1950.78  5010.6 1951.28
  5043.8 1953.02    5100 1953.45  5107.3 1954.38  5170.9 1952.37  5193.8 1952.85
  5200.1 1951.89  5214.7 1952.72  5220.9 1951.71  5229.3 1952.58  5235.5  1951.5
  5264.7 1953.03  5285.5 1952.72  5329.3  1956.3  5409.5 1958.01    5421 1959.87
  5507.9 1963.72  5587.3 1963.88  5595.3 1965.02  5616.4 1965.58  5756.8 1967.78
#Mann= 6 ,-1 , 0
  4442.2     .12       0  4804.2     .05       0  4889.9     .12       0
  5004.8     .07       0  5010.6     .12       0  5409.5     .05       0
Bank Sta=5004.8,5010.6
XS Rating Curve= 0 ,0
Exp/Cntr=0.3,0.1

Type RM Length L Ch R = 1 ,39771   ,683,683,683
BEGIN DESCRIPTION:
Elm 01 91 39771.35
END DESCRIPTION:
XS GIS Cut Line= 3
      1604077.78      6788124.77      1604464.05      6787894.75
      1605186.66      6787478.11
#Sta/Elev= 30
  4550.3 1954.04  4677.2 1954.96  4802.6 1954.85  4808.4 1955.76    4824 1954.64
  4884.4 1954.13  4946.6  1949.1  4962.2 1946.79  5026.6 1947.42  5098.4 1945.21
  5098.9 1944.71  5104.2 1945.21  5122.8 1945.48  5128.6 1946.95  5138.6 1946.78
  5144.4 1947.97  5160.2 1945.99  5174.1 1946.19  5246.4 1949.56  5279.2 1946.78
  5305.3 1947.23  5312.6 1945.95  5348.4 1947.49  5379.9 1945.37  5402.4 1947.18
  5480.7 1950.38    5532 1953.33  5642.8 1956.71  5811.2 1959.08    5834  1959.2
#Mann= 9 ,-1 , 0
  4550.3     .12       0  4677.2     .05       0  4884.4     .12       0
  5098.4     .07       0  5104.2     .12       0  5279.2     .05       0
  5402.4     .12       0  5480.7     .05       0  5811.2     .12       0
Bank Sta=5098.4,5104.2
XS Rating Curve= 0 ,0
Exp/Cntr=0.3,0.1

Type RM Length L Ch R = 1 ,39088   ,252,252,252
BEGIN DESCRIPTION:
Elm 01 91 39088.03
END DESCRIPTION:
XS GIS Cut Line= 3
       1604214.5      6788228.95      1604856.84      6788254.99
      1605586.01      6788103.08
#Sta/Elev= 30
  4359.4 1952.81  4445.2 1952.51  4590.1 1950.89  4680.2 1948.83  4706.8 1947.62
  4720.2 1946.78  4740.2 1946.67  4760.2 1945.07  4780.2 1944.42  4850.3 1943.29
  4900.3 1941.65  4954.3 1941.63  4970.4  1940.4  4990.4 1940.41  4995.6 1938.58
  4996.1 1938.08  5002.1 1938.58  5008.8 1940.05  5041.2 1942.77  5063.9 1943.41
  5143.4 1942.39  5217.8 1945.95  5235.3 1947.01    5259 1947.02  5341.4 1949.92
  5378.3 1951.45  5523.2 1953.35  5644.7 1955.07  5658.2 1955.27  5747.1 1956.52
#Mann= 10 ,-1 , 0
  4359.4     .12       0  4445.2     .05       0  4706.8     .12       0
  4995.6     .07       0  5002.1     .12       0  5217.8     .05       0
  5341.4     .12       0  5523.2     .05       0  5644.7     .12       0
  5658.2     .05       0
Bank Sta=4995.6,5002.1
XS Rating Curve= 0 ,0
Exp/Cntr=0.3,0.1

Type RM Length L Ch R = 1 ,38836   ,135,135,135
BEGIN DESCRIPTION:
Elm 01 91 38835.62
END DESCRIPTION:
XS GIS Cut Line= 3
      1603697.79      6788452.29      1604754.67      6788460.97
      1605461.05       6788413.3
#Sta/Elev= 30
  3943.3 1952.29  3980.5 1951.41  4040.5 1951.29  4190.5 1947.53  4210.5 1947.65
  4240.5  1945.5  4360.5 1945.75  4430.5 1947.91  4520.5 1949.34  4600.5 1949.94
  4650.5 1948.65  4690.5 1949.01  4720.5 1948.15  4830.5 1947.04  4900.5 1944.17
  4950.5 1941.28  5017.3 1939.07  5017.8 1938.57  5023.3 1938.57  5023.8 1939.07
  5050.7 1940.14  5070.7 1942.16  5090.8 1941.79  5100.8 1940.95  5229.7 1941.27
  5428.5 1947.01  5461.6 1948.34  5527.9 1949.18  5627.3 1950.73  5708.2 1951.51
#Mann= 7 ,-1 , 0
  3943.3     .12       0  5017.3     .07       0  5023.8     .12       0
  5229.7     .05       0  5428.5     .12       0  5527.9     .05       0
  5627.3     .12       0
Bank Sta=5017.3,5023.8
XS Rating Curve= 0 ,0
Exp/Cntr=0.3,0.1

Type RM Length L Ch R = 1 ,38701   ,189,189,189
BEGIN DESCRIPTION:
Elm 01 91 38701.06
END DESCRIPTION:
XS GIS Cut Line= 3
       1603667.4      6788634.59       1604752.5      6788595.52
      1605329.78      6788599.86
#Sta/Elev= 30
  3912.8 1952.06  4030.5 1951.48  4260.6 1948.03  4380.7 1943.36  4400.7 1940.99
  4410.7 1941.03  4430.7 1942.95  4480.8 1943.24  4514.3  1945.2  4541.6 1945.78
  4590.8 1946.87  4640.9 1946.92    4841 1945.31    4851 1944.34  4921.1 1943.46
  4951.1 1941.68  4961.1 1940.51  4977.8 1936.83  4978.3 1936.33  4984.3 1936.83
  4991.1 1937.22  4997.4 1938.66  5041.1 1939.08  5071.1 1941.04  5111.1 1939.62
  5141.1 1940.55  5224.7 1940.53  5321.1 1941.47  5471.1 1945.28  5575.9 1946.54
#Mann= 5 ,-1 , 0
  3912.8     .05       0  4541.6     .12       0  4977.8     .07       0
  4984.3     .12       0  5224.7     .05       0
Bank Sta=4977.8,4984.3
XS Rating Curve= 0 ,0
Exp/Cntr=0.3,0.1

Type RM Length L Ch R = 1 ,38512   ,443,443,443
BEGIN DESCRIPTION:
Elm 01 91 38512.37
END DESCRIPTION:
XS GIS Cut Line= 3
      1603754.26       6789046.9      1604726.45      6788760.45
      1605314.52      6788669.31
#Sta/Elev= 30
  3984.8  1953.3  4016.8 1952.56  4027.3 1953.25  4033.2 1952.04  4110.7  1950.2
    4354 1946.65  4444.3 1944.61  4459.2 1944.06  4506.8 1940.12  4538.1 1939.34
  4558.9 1939.16  4579.8 1940.52  4590.2  1940.1    4706 1942.74  4741.5 1942.23
    4757 1942.99  4861.3  1943.2  4951.9 1940.62  4981.9 1937.21  4982.4 1936.71
  4988.5 1937.21  5077.8 1938.06  5118.3 1937.41  5175.7 1938.86    5217 1938.39
  5229.6 1938.15  5259.9 1939.29  5300.4 1938.97  5361.1 1939.73  5593.4 1945.72
#Mann= 5 ,-1 , 0
  3984.8     .05       0    4706     .12       0  4981.9     .07       0
  4988.5     .12       0    5217     .05       0
Bank Sta=4981.9,4988.5
XS Rating Curve= 0 ,0
Exp/Cntr=0.3,0.1

Type RM Length L Ch R = 1 ,38069   ,305,305,305
BEGIN DESCRIPTION:
Elm 01 91 38068.87
END DESCRIPTION:
XS GIS Cut Line= 3
      1604576.75      6789370.23      1604871.85      6789055.59
      1605291.43      6788817.69
#Sta/Elev= 30
  4566.2 1941.64  4707.9  1941.5    4807 1938.58  4828.5 1938.89    4892 1937.47
  4920.3 1936.54  4927.2 1935.58  4947.6 1935.54  4962.8 1934.79    4977 1932.47
    4980 1930.96  4980.5 1930.46  4987.2 1930.46  4987.7 1930.96  4996.2 1932.46
  5000.2 1932.46  5012.7 1934.97  5035.7 1936.41  5058.3 1937.08  5117.3 1936.55
  5173.6 1935.57  5219.6 1935.67  5231.3 1936.46  5277.1 1936.77  5371.3 1940.09
  5403.1  1940.4    5438 1942.27  5452.1  1945.2    5461 1947.82  5479.9 1949.18
#Mann= 5 ,-1 , 0
  4566.2     .05       0  4947.6     .12       0    4980     .07       0
  4987.7     .12       0  5117.3     .05       0
Bank Sta=4980,4987.7
XS Rating Curve= 0 ,0
Exp/Cntr=0.3,0.1

Type RM Length L Ch R = 1 ,37764   ,517,517,517
BEGIN DESCRIPTION:
Elm 01 91 37764.1
END DESCRIPTION:
XS GIS Cut Line= 3
      1604658.86       6789622.6       1605021.3      6789303.57
      1605316.41      6789023.65
#Sta/Elev= 30
    4518    1939    4823 1938.15  4922.6 1936.29  4951.1 1937.77  4963.2 1936.42
  4979.1 1934.38  4992.8 1930.26    5000 1929.55  5003.4 1927.94  5003.9 1927.44
  5010.6 1927.44  5011.1 1927.94  5021.4  1933.2  5028.7 1934.04  5071.1  1934.4
  5113.6 1932.84  5120.5 1933.38  5127.8 1932.98  5134.7 1934.38  5170.2 1933.59
  5177.1 1934.07  5184.4  1933.5  5232.9 1933.66  5276.2 1933.43  5361.2 1935.57
  5375.3 1934.42  5382.2 1935.35  5389.5 1935.31  5403.2  1939.5  5407.6  1939.5
#Mann= 5 ,-1 , 0
    4518     .05       0  4963.2     .12       0  5003.4     .07       0
  5011.1     .12       0  5232.9     .05       0
Bank Sta=5003.4,5011.1
XS Rating Curve= 0 ,0
Exp/Cntr=0.3,0.1

Type RM Length L Ch R = 1 ,37247   ,399,399,399
BEGIN DESCRIPTION:
Elm 01 91 37246.55
END DESCRIPTION:
XS GIS Cut Line= 3
      1604550.37      6789822.23      1605403.25      6789561.81
      1605974.04      6789401.21
#Sta/Elev= 30
  4106.2 1937.61  4351.5 1937.26    4592 1932.91  4683.3 1929.37  4811.6 1929.21
  4874.3 1931.28  4966.3 1929.16    4989 1928.77  4992.4 1926.51  4992.9 1926.01
  5000.1 1926.51  5028.1 1928.92  5145.8 1927.11  5174.7 1931.71  5179.9  1930.9
  5213.9 1940.96  5219.1 1940.29  5238.7 1947.39  5296.1 1953.85    5353 1957.61
  5373.7 1954.51  5384.1 1954.75  5394.5 1957.42  5399.7 1956.29  5433.7 1966.91
  5438.9 1965.12  5446.5 1968.19    5473  1971.5  5546.3 1975.76  5590.9 1974.38
#Mann= 5 ,-1 , 0
  4106.2     .05       0  4966.3     .12       0  4992.4     .07       0
  5000.1     .12       0  5296.1     .05       0
Bank Sta=4992.4,5000.1
XS Rating Curve= 0 ,0
Exp/Cntr=0.3,0.1

Type RM Length L Ch R = 1 ,36848   ,130,130,130
BEGIN DESCRIPTION:
Elm 01 91 36847.94
END DESCRIPTION:
XS GIS Cut Line= 4
       1604923.6      6789818.61      1605405.42      6789885.89
      1605505.24      6789929.29      1605750.24      6789907.61
#Sta/Elev= 30
  4404.7 1933.68    4439 1932.54  4456.6 1933.07  4476.8  1930.8  4608.1 1926.79
  4688.8 1926.46  4724.9 1925.75  4769.6 1926.26  4860.5 1925.53  4908.1 1926.12
  4923.4 1925.27    4937 1922.64  4945.3 1921.85  4960.4  1919.2  4979.8  1918.8
  4980.3  1918.3  4987.4  1918.3  4987.9  1918.8    5050 1918.88  5059.5 1920.84
  5080.1 1926.41  5099.1 1929.11  5110.2  1931.9  5120.3 1936.93  5130.3 1942.72
  5140.3 1946.25  5150.4 1948.33  5160.4 1949.12  5200.6 1950.19    5246 1949.58
#Mann= 5 ,-1 , 0
  4404.7     .05       0  4979.8     .05       0  4987.9     .05       0
  5059.5     .12       0  5099.1     .05       0
Bank Sta=4979.8,4987.9
XS Rating Curve= 0 ,0
Exp/Cntr=0.3,0.1

Type RM Length L Ch R = 1 ,36718   ,329,329,329
BEGIN DESCRIPTION:
Elm 01 91 36718.14
END DESCRIPTION:
XS GIS Cut Line= 5
      1604862.87      6789901.08       1605312.1       6789957.5
      1605453.16      6790039.97      1605533.46      6790074.69
      1605806.87      6789996.57
#Sta/Elev= 30
  4383.9 1934.93  4480.7 1932.35  4486.8 1931.06  4537.2 1928.89  4678.3  1925.7
  4738.8 1925.81  4754.9 1922.64  4755.4 1922.14    4763 1922.64    4769 1926.02
  4868.2  1926.3  4905.4    1929  4985.5 1929.58  4991.3 1930.86  5007.6  1930.3
  5013.1 1931.63  5067.4 1933.06  5090.6  1933.4  5099.5 1931.63  5127.8 1931.22
    5133 1930.11  5161.6 1931.76  5166.8 1930.72  5193.1 1933.91  5234.4 1935.69
  5245.1 1938.73  5286.7 1941.16  5307.2    1941  5312.4  1942.1  5371.9 1942.99
#Mann= 3 ,-1 , 0
  4383.9     .05       0  4754.9     .05       0    4763     .05       0
Bank Sta=4754.9,4763
XS Rating Curve= 0 ,0
Exp/Cntr=0.3,0.1

Type RM Length L Ch R = 1 ,36389   ,380,380,380
BEGIN DESCRIPTION:
Elm 01 91 36389.27
END DESCRIPTION:
XS GIS Cut Line= 4
      1604832.47      6790018.25      1605160.19      6790135.45
       1605479.2      6790198.39      1605835.09      6790087.71
#Sta/Elev= 30
  4651.9 1935.14  4668.3 1935.35  4718.3 1932.96  4729.8 1933.23  4739.5 1931.19
    4750 1930.47    4867 1926.74  4888.2 1925.14  4929.3 1925.01  4934.6 1923.88
  4951.9 1923.49  4992.2 1920.18  4992.7 1919.68  5000.3 1920.18  5004.9 1921.44
    5015 1921.57  5290.2 1923.34  5339.8 1924.54  5447.9 1925.04  5467.3 1926.04
  5480.5 1924.95  5498.7 1925.17  5507.8 1926.67    5513 1926.01  5519.7  1927.3
  5545.6 1928.36  5561.6 1931.72  5578.1 1933.31  5667.9 1936.78  5697.8 1938.65
#Mann= 4 ,-1 , 0
  4651.9     .05       0  4992.2     .05       0  5000.3     .05       0
  5667.9     .12       0
Bank Sta=4992.2,5000.3
XS Rating Curve= 0 ,0
Exp/Cntr=0.3,0.1

Type RM Length L Ch R = 1 ,36009   ,561,561,561
BEGIN DESCRIPTION:
Elm 01 91 36008.85
END DESCRIPTION:
XS GIS Cut Line= 3
       1604419.6      6790358.07      1605124.93      6790468.75
       1605631.4      6790481.74
#Sta/Elev= 30
  4286.3 1940.26  4317.6 1937.55  4332.3 1937.31  4380.2 1934.34  4413.2 1934.03
  4554.9 1928.16  4656.2 1925.93  4676.4 1926.19  4686.5 1925.05  4703.4 1921.64
    4727 1920.33  4766.1 1920.62  4868.7 1918.15  4896.4 1919.34  4980.1 1919.33
  5006.2 1916.96  5006.7 1916.46  5014.4 1916.96  5050.3 1922.57  5080.4 1923.27
  5100.4  1925.7  5110.4 1926.15  5200.4 1928.77  5240.4 1928.26  5260.4 1928.88
  5270.4 1928.14  5310.4 1928.24  5320.4 1927.62  5350.4 1928.39  5506.9 1927.31
#Mann= 3 ,-1 , 0
  4286.3     .05       0  5006.2     .05       0  5014.4     .05       0
Bank Sta=5006.2,5014.4
XS Rating Curve= 0 ,0
Exp/Cntr=0.3,0.1

Type RM Length L Ch R = 1 ,35448   ,339,339,339
BEGIN DESCRIPTION:
Elm 01 91 35448.38
END DESCRIPTION:
XS GIS Cut Line= 3
      1604395.72      6790776.91      1605012.08       6790792.1
      1605539.45      6790748.69
#Sta/Elev= 30
  4386.6 1933.54  4405.9 1933.68  4465.9 1931.88  4555.9 1930.31    4716 1928.64
    4756 1928.69    4776 1927.11    4856 1924.25    4906 1920.63    4916 1920.35
    4946 1917.11  4966.1 1916.38  4996.1  1916.8  5016.1 1916.33  5026.1 1917.44
  5046.2 1917.58  5056.2 1915.69  5062.1 1913.69  5062.6 1913.19  5069.9 1913.19
  5070.4 1913.69  5076.3 1916.69  5086.3 1917.34  5112.8  1916.9  5186.7 1921.13
  5206.8 1921.33  5246.9 1922.85  5467.6 1926.25  5476.2 1925.85  5532.3 1925.93
#Mann= 3 ,-1 , 0
  4386.6     .05       0  5062.1     .05       0  5070.4     .05       0
Bank Sta=5062.1,5070.4
XS Rating Curve= 0 ,0
Exp/Cntr=0.3,0.1

Type RM Length L Ch R = 1 ,35109   ,505,505,505
BEGIN DESCRIPTION:
Elm 01 91 35108.69
END DESCRIPTION:
XS GIS Cut Line= 3
      1604337.16      6791052.52      1605051.14       6791061.2
      1605765.69       6790842.5
#Sta/Elev= 30
  4283.5 1931.35  4411.3 1928.57  4661.4 1926.74  4741.4 1926.82  4761.4 1925.58
  4771.4 1926.05  4841.4 1924.93  4881.4 1923.36  4911.4 1921.43  4931.4 1918.94
  4961.4 1917.14  4971.4 1915.31    4997 1912.97  5021.4 1912.96  5026.6 1914.61
  5059.4 1914.32  5064.6 1915.17  5221.2 1914.46  5242.1 1915.47  5261.3 1912.41
  5279.8 1912.37  5280.3 1911.87  5287.6 1911.87  5288.1 1912.37    5294 1914.73
  5299.3 1917.76  5304.8 1918.37  5402.8 1921.68  5555.8 1924.47  5744.8 1924.63
#Mann= 3 ,-1 , 0
  4283.5     .05       0  5279.8     .05       0  5288.1     .05       0
Bank Sta=5279.8,5288.1
XS Rating Curve= 0 ,0
Exp/Cntr=0.3,0.1

Type RM Length L Ch R = 1 ,34604   ,502,502,502
BEGIN DESCRIPTION:
Elm 01 91 34603.91
END DESCRIPTION:
XS GIS Cut Line= 3
      1604469.51      6791223.96      1605400.53      6791191.41
      1605736.04      6791213.05
#Sta/Elev= 30
  4070.2 1928.27  4094.2 1926.78  4105.7 1927.05  4115.7 1926.55  4175.8 1925.77
  4387.4 1924.86  4405.9 1924.11    4546 1923.12    4656    1920  4696.1 1917.92
  4716.1 1917.39  4786.1 1913.41  4826.2 1913.04  4886.2 1913.62  4936.2 1913.01
  4966.2 1913.34  4986.3 1912.91  4996.3 1911.78  4997.3 1911.15  4997.8 1910.65
  5005.2 1910.65  5005.7 1911.15  5028.9 1911.16  5046.4 1914.99  5066.4    1918
  5076.4 1919.01  5096.5 1919.65  5176.6 1921.06  5286.9 1921.45    5338 1920.96
#Mann= 3 ,-1 , 0
  4070.2     .05       0  4997.3     .05       0  5005.7     .05       0
Bank Sta=4997.3,5005.7
XS Rating Curve= 0 ,0
Exp/Cntr=0.3,0.1

Type RM Length L Ch R = 1 ,34102   ,500,500,500
BEGIN DESCRIPTION:
Elm 01 91 34101.95
END DESCRIPTION:
XS GIS Cut Line= 3
      1604695.29      6791506.86      1605406.18      6791558.94
      1606081.64      6791397.87
#Sta/Elev= 30
  4287.8 1921.73  4337.6 1922.39    4468 1921.01  4608.4 1914.47  4649.5 1913.25
    4849 1912.05  4889.1 1910.64  4909.2 1909.39  4921.8 1907.72  4939.3 1909.19
  4959.3 1909.31  4969.3 1908.05  5005.5 1906.68    5006 1906.18  5013.9 1906.68
  5030.8 1909.09  5072.9 1910.29  5109.9 1910.39    5133 1907.61  5143.3 1907.84
  5163.9 1912.47  5174.2 1913.58    5205 1916.46  5241.4 1917.86  5372.9 1917.27
  5400.3 1915.78  5472.3 1916.98  5583.4 1915.39  5630.7  1916.5    5695 1916.71
#Mann= 3 ,-1 , 0
  4287.8     .05       0  5005.5     .05       0  5013.9     .05       0
Bank Sta=5005.5,5013.9
XS Rating Curve= 0 ,0
Exp/Cntr=0.3,0.1

Type RM Length L Ch R = 1 ,33602   ,523,523,523
BEGIN DESCRIPTION:
Elm 01 91 33602.16
END DESCRIPTION:
XS GIS Cut Line= 3
      1604903.61       6791845.4      1605104.09      6791855.82
      1605950.24      6791590.25
#Sta/Elev= 30
    4799 1920.78  4802.2 1920.78  4810.4 1918.93  4820.4 1914.78  4830.4  1912.6
  4840.4 1911.93  4900.5 1912.53  4930.6 1909.07  4940.5 1908.44  4945.5 1909.47
  4950.6 1909.19  4976.4 1903.31  4976.9 1902.81  4984.8 1903.31  4990.7 1904.28
  5002.9 1904.52  5007.6 1905.51    5095 1907.44  5104.8 1906.79  5168.4  1906.8
  5174.9 1906.23  5277.4  1907.8  5379.9 1911.73  5412.3 1911.35  5439.5 1913.07
  5444.7 1912.42  5461.9    1914  5509.6 1915.39  5671.5 1914.78  5886.6 1912.43
#Mann= 3 ,-1 , 0
    4799     .05       0  4976.4     .05       0  4984.8     .05       0
Bank Sta=4976.4,4984.8
XS Rating Curve= 0 ,0
Exp/Cntr=0.3,0.1

Type RM Length L Ch R = 1 ,33079   ,1126,1126,1126
BEGIN DESCRIPTION:
Elm 01 91 33078.68
END DESCRIPTION:
XS GIS Cut Line= 3
      1604742.11      6792267.27      1605455.66       6792160.5
      1606377.52      6791879.26
#Sta/Elev= 30
  4279.4 1924.59    4343  1924.1  4353.1 1923.27  4377.1  1923.7  4474.4 1919.41
  4504.8 1918.81    4525 1917.18  4535.1 1917.43  4545.2 1916.51  4585.7 1910.02
  4605.9 1908.29  4666.6 1904.78  4743.2    1902  4743.7  1901.5  4751.7    1902
  4787.9 1902.23  4818.2 1904.02  4851.2 1904.35  4969.9 1903.43  4990.1 1902.08
  5003.2 1902.45  5031.7 1906.08  5073.4 1906.83    5201 1906.05  5299.5 1904.54
    5436 1904.84  5605.3 1907.25  5648.5 1909.16  5817.9 1910.34  5964.7 1912.98
#Mann= 3 ,-1 , 0
  4279.4     .05       0  4743.2     .03       0  4751.7     .05       0
Bank Sta=4743.2,4751.7
XS Rating Curve= 0 ,0
Exp/Cntr=0.3,0.1

Type RM Length L Ch R = 1 ,31953   ,369,369,369
BEGIN DESCRIPTION:
Mapping XS b4a205c2
END DESCRIPTION:
XS GIS Cut Line= 4
      1604834.34      6792713.14      1605580.85      6792656.71
      1606600.82      6792300.81      1606851.28      6792141.03
#Sta/Elev= 30
  3852.1 1923.36  3892.9 1922.53  3912.9 1923.02    3953 1920.89  4003.2 1920.46
  4033.3 1917.25  4073.4 1916.12  4083.4 1914.64  4133.6 1912.16  4163.6 1907.83
  4173.7 1907.08  4250.4 1903.26  4381.9 1900.63  4574.8 1902.34  4668.1 1900.71
  4774.6 1900.43  4885.5  1899.1  4922.9 1897.94  4965.2 1898.35    4997 1897.35
  5004.5 1895.55    5005 1895.05    5015 1895.55  5018.2 1897.74  5040.8 1904.35
  5066.6  1905.3  5159.8 1904.78  5185.5 1905.92  5325.3  1907.6  5978.1 1912.74
#Mann= 3 ,-1 , 0
  3852.1     .05       0  5004.5     .05       0    5015     .05       0
Bank Sta=5004.5,5015
XS Rating Curve= 0 ,0
Exp/Cntr=0.3,0.1

Type RM Length L Ch R = 1 ,31584   ,1709,1709,1709
BEGIN DESCRIPTION:
Mapping XS 77559c60
END DESCRIPTION:
XS GIS Cut Line= 4
       1604834.3        6792839.      1605220.61      6792891.09
      1605546.13      6792865.05      1607208.42      6792769.56
#Sta/Elev= 30
  3914.2 1923.14  3965.4 1921.17  4066.3  1920.3  4092.6 1918.42  4288.3 1914.29
  4388.7 1909.51  4428.8 1909.25  4519.1 1898.69  4579.3 1895.08  4670.4 1898.95
  4889.9 1899.32    4950 1898.75    4960 1896.82  4964.6 1894.56  4965.1 1894.06
  4975.3 1894.56    4990 1896.48  5050.1 1898.58  5130.3 1898.67  5180.3  1901.1
  5270.5  1903.1  5320.6 1900.92  5330.6  1902.4  5380.7 1903.69  5821.4 1905.65
  6051.8 1905.37  6236.4 1907.74  6252.1 1910.55  6272.1 1909.53  6295.6 1910.31
#Mann= 3 ,-1 , 0
  3914.2     .05       0  4964.6     .05       0  4975.3     .05       0
Bank Sta=4964.6,4975.3
XS Rating Curve= 0 ,0
Exp/Cntr=0.3,0.1

Type RM Length L Ch R = 1 ,29875   ,424,424,424
BEGIN DESCRIPTION:
Elm 01 91 29875.16
END DESCRIPTION:
XS GIS Cut Line= 3
      1604759.65      6792913.17      1605204.48      6793171.39
      1606165.89      6793637.98
#Sta/Elev= 30
    4486 1921.42  4501.8 1921.99  4550.6  1920.9  4677.2 1920.39    4727 1918.46
  4764.2 1918.64    4770 1918.05  4815.9 1917.75  4919.1 1915.46  4931.6  1914.2
  4940.6 1908.75  4946.4 1907.83  4962.1 1897.15  4967.9 1896.06  4983.6  1888.7
  4992.3 1888.28  4992.8 1887.78  5002.7 1887.78  5003.2 1888.28    5012 1890.06
  5050.4 1890.37  5056.5  1891.7  5118.1 1892.31  5156.5  1893.1  5168.8 1894.22
  5185.8 1893.95  5276.1 1895.73    5417 1894.72  5656.7 1897.09    6069 1896.53
#Mann= 3 ,-1 , 0
    4486     .05       0  4992.3     .05       0  5003.2     .05       0
Bank Sta=4992.3,5003.2
XS Rating Curve= 0 ,0
Exp/Cntr=0.3,0.1

Type RM Length L Ch R = 1 ,29451   ,336,336,336
BEGIN DESCRIPTION:
Elm 01 91 29450.78
END DESCRIPTION:
XS GIS Cut Line= 3
      1604462.31      6793577.42      1605108.13      6793548.78
       1606006.6       6793624.3
#Sta/Elev= 30
  4357.2 1921.27  4399.9 1919.61    4440 1916.41    4456 1916.94    4461  1915.2
  4520.1 1913.99  4560.1 1908.62  4610.1 1903.47  4670.2 1893.52  4740.3 1891.63
  4840.4 1890.03  4906.9 1889.77  4960.5 1888.61    4985 1887.07  4985.5 1886.57
  4995.5 1886.57    4996 1887.07  5020.6 1889.13  5054.9 1889.62  5110.9 1888.97
    5151 1890.08  5221.3 1890.78  5261.4 1892.34  5281.5 1892.14  5311.6 1893.12
  5442.1 1893.46  5654.4 1896.32  5692.9 1895.65  5723.1 1896.13  5905.3 1896.08
#Mann= 3 ,-1 , 0
  4357.2     .05       0    4985     .05       0    4996     .05       0
Bank Sta=4985,4996
XS Rating Curve= 0 ,0
Exp/Cntr=0.3,0.1

Type RM Length L Ch R = 1 ,29115   ,185,185,185
BEGIN DESCRIPTION:
Elm 01 91 29115.08
END DESCRIPTION:
XS GIS Cut Line= 3
      1604365.98      6793809.19      1605303.44       6793751.9
      1606097.69      6793728.47
#Sta/Elev= 30
  4059.7 1927.36  4078.8 1927.19  4157.5 1922.92  4162.6 1924.01  4249.1 1917.19
  4259.1 1915.42  4279.1 1914.12  4324.7 1908.63  4339.2 1909.67  4369.3 1905.43
  4409.4 1901.78  4429.4  1898.6  4519.6 1892.83  4689.9 1888.16  4821.1 1887.52
  4870.2 1888.87  4920.3 1888.93    5005 1887.04  5005.5 1886.54    5016 1887.04
  5080.5 1892.61  5200.6  1893.2  5303.2 1894.84  5460.7 1895.13  5550.7 1895.95
  5560.7 1896.69  5590.7 1895.62  5637.7 1896.29  5660.8 1895.68  5793.5 1895.94
#Mann= 3 ,-1 , 0
  4059.7     .05       0    5005     .03       0    5016     .05       0
Bank Sta=5005,5016
XS Rating Curve= 0 ,0
Exp/Cntr=0.3,0.1
