HEC-RAS study Elm 01 91.prj: Elm 01 91 Base Level Engineering

--- Elm 01 91.g01 (geometry) --- (continued)

Type RM Length L Ch R = 1 ,28930   ,441,441,441
BEGIN DESCRIPTION:
Elm 01 91 28929.57
END DESCRIPTION:
XS GIS Cut Line= 3
      1604490.98      6794007.11       1605274.8      6793923.78
       1606041.5      6793908.18
#Sta/Elev= 30
  4218.3 1923.96  4272.6 1924.79  4312.9 1928.47    4333 1927.57  4354.9 1925.02
  4423.5 1911.43  4442.4 1908.94    4514 1903.64    4524 1902.16    4540  1896.9
    4545 1897.15  4564.3 1893.08  4588.2 1890.58  4752.3 1888.21  4915.2 1886.72
  4926.3 1885.69  4930.8 1882.63  4931.3 1882.13  4941.8 1882.63  4946.4 1886.66
  4956.5 1886.86  5026.7 1885.84  5036.7 1884.32  5043.2 1886.22  5048.2 1885.64
  5056.7  1889.2  5066.8 1890.13  5116.8 1889.19  5326.8 1892.53  5773.4 1894.36
#Mann= 5 ,-1 , 0
  4218.3     .05       0  4588.2     .12       0  4752.3     .05       0
  4930.8     .05       0  4941.8     .05       0
Bank Sta=4930.8,4941.8
XS Rating Curve= 0 ,0
Exp/Cntr=0.3,0.1

Type RM Length L Ch R = 1 ,28489   ,471,471,471
BEGIN DESCRIPTION:
Elm 01 91 28488.88
END DESCRIPTION:
XS GIS Cut Line= 3
      1604563.87      6794264.92       1605346.7      6794285.66
      1606870.44      6794272.74
#Sta/Elev= 30
  4216.9 1921.49    4258 1921.35    4278 1922.14  4318.1 1926.04  4358.1 1924.61
  4368.1 1922.56  4398.1 1913.23  4438.1 1899.71  4458.1 1891.81  4468.1 1888.98
  4478.1 1887.59  4508.1 1887.69  4548.1 1886.37  4708.2 1886.14  4818.2  1884.8
  4938.3  1885.5  4958.3 1884.08  4978.3 1884.75    5000 1883.78  5002.7  1882.5
  5003.2    1882  5013.9  1882.5  5018.3 1882.52  5038.3 1886.12  5168.3 1888.62
  5408.3 1889.65  5678.3  1889.4  5868.3 1890.83  6338.4 1897.31  6523.8 1897.54
#Mann= 3 ,-1 , 0
  4216.9     .05       0  5002.7     .05       0  5013.9     .05       0
Bank Sta=5002.7,5013.9
XS Rating Curve= 0 ,0
Exp/Cntr=0.3,0.1

Type RM Length L Ch R = 1 ,28018   ,787,787,787
BEGIN DESCRIPTION:
Elm 01 91 28018.96
END DESCRIPTION:
XS GIS Cut Line= 3
       1604501.4      6794582.63      1605254.83      6794579.16
      1606870.38      6794585.23
#Sta/Elev= 30
    4243 1924.06  4346.6 1925.48  4386.6 1924.56  4396.6 1923.37  4436.6 1914.29
  4516.6 1904.63  4556.6  1894.9  4606.6 1887.93  4626.6 1887.05  4656.6 1889.81
  4736.6 1884.07  4786.6    1883  4956.6 1883.91  4988.4 1880.23  4988.9 1879.73
  4999.7 1880.23  5016.6 1881.05  5036.6 1883.92  5056.6 1884.62  5136.6 1884.13
  5196.6  1885.6  5346.6 1886.44  5426.6  1885.5  5486.6  1886.3  5496.6 1887.77
  5576.6  1887.8  5626.6 1889.19  5966.6  1892.8  6396.6 1895.53    6612 1895.64
#Mann= 3 ,-1 , 0
    4243     .05       0  4988.4     .05       0  4999.7     .05       0
Bank Sta=4988.4,4999.7
XS Rating Curve= 0 ,0
Exp/Cntr=0.3,0.1

Type RM Length L Ch R = 1 ,27231   ,995,995,995
BEGIN DESCRIPTION:
Elm 01 91 27231.12
END DESCRIPTION:
XS GIS Cut Line= 3
      1604583.44      6794777.93      1604989.73      6794949.82
      1606384.92      6795363.56
#Sta/Elev= 30
  4556.3  1908.6  4566.4 1908.96  4595.5 1905.97  4619.2 1905.38  4624.6 1903.65
  4642.9 1903.21  4648.3 1901.17  4666.6 1900.66  4677.4 1897.84  4772.2 1888.25
  4830.4 1884.91  4916.3 1881.63  4959.7 1881.02  4970.6 1880.17    4978 1878.24
  4997.3  1877.5  4997.8    1877  5008.7  1877.5  5013.6 1879.63  5046.9 1881.21
  5179.8 1882.43  5232.4 1882.24  5263.7 1879.51  5328.4 1878.29  5388.9 1882.34
  5499.7 1883.98  5609.9 1884.26  5886.2 1887.44  6247.2 1888.23  6452.7 1888.99
#Mann= 4 ,-1 , 0
  4556.3     .05       0  4997.3     .05       0  5008.7     .05       0
  6247.2     .12       0
Bank Sta=4997.3,5008.7
XS Rating Curve= 0 ,0
Exp/Cntr=0.3,0.1

Type RM Length L Ch R = 1 ,26236   ,563,563,563
BEGIN DESCRIPTION:
Elm 01 91 26235.65
END DESCRIPTION:
XS GIS Cut Line= 3
      1603943.05      6795514.09      1604993.42       6795644.3
      1606120.98       6795609.6
#Sta/Elev= 30
  3939.7 1894.26  4040.3 1891.99  4153.3 1890.01    4385 1882.07  4445.5  1878.1
  4475.7 1874.98  4505.9 1874.78  4556.3  1876.4  4576.3 1876.18  4581.3  1875.3
  4743.2 1876.48  4898.9 1875.76  4969.5 1876.31  4979.5 1874.22  4980.4  1869.4
  4980.9  1868.9  4991.8  1869.4  5029.7 1872.36  5069.7 1873.37  5109.7 1875.48
  5199.8 1877.32  5229.8 1878.89  5279.8 1878.52  5379.9 1879.73  5439.9 1878.93
  5479.9 1881.16  5509.9 1880.29    5580 1880.67  5692.8 1882.49  6126.2 1885.47
#Mann= 4 ,-1 , 0
  3939.7     .12       0  4040.3     .05       0  4980.4     .05       0
  4991.8     .05       0
Bank Sta=4980.4,4991.8
XS Rating Curve= 0 ,0
Exp/Cntr=0.3,0.1

Type RM Length L Ch R = 1 ,25673   ,574,574,574
BEGIN DESCRIPTION:
Elm 01 91 25672.7
END DESCRIPTION:
XS GIS Cut Line= 3
      1603847.62      6796165.13      1604750.36      6796082.67
      1606147.93      6795900.38
#Sta/Elev= 30
  4094.2 1914.18  4161.9  1913.5  4181.9 1914.13  4272.3 1911.13  4332.5 1906.87
  4342.6 1904.38  4372.7 1902.22  4523.4 1893.56  4603.7 1887.53  4834.6 1877.95
  4883.5 1873.59  4888.5 1873.86  4894.9 1872.22  4904.9 1871.16  5009.5 1867.59
    5010 1867.09  5021.5 1867.59  5065.9 1869.85  5073.2  1868.9  5078.2 1869.55
  5096.1 1868.44  5126.4 1868.13  5166.7 1870.96  5217.2 1870.32  5509.6  1875.9
  5590.3 1875.84  5731.5 1877.61  5953.3 1878.67  6054.2 1880.59  6410.1 1884.47
#Mann= 3 ,-1 , 0
  4094.2     .05       0  5009.5     .05       0  5021.5     .05       0
Bank Sta=5009.5,5021.5
XS Rating Curve= 0 ,0
Exp/Cntr=0.3,0.1

Type RM Length L Ch R = 1 ,25099   ,452,452,452
BEGIN DESCRIPTION:
Elm 01 91 25099.02
END DESCRIPTION:
XS GIS Cut Line= 3
      1604003.87      6796590.47      1605158.35      6796442.91
      1606516.81      6796199.86
#Sta/Elev= 30
  3831.6 1902.48  3992.1 1897.35  4043.9 1894.58  4048.9 1895.09    4115 1889.67
  4192.4 1886.02  4283.1 1880.96  4292.6 1881.14  4362.9 1877.65    4488 1873.82
    4609 1871.94  4810.6 1871.06  4871.1 1868.21  4911.1 1868.39  4931.6 1866.41
  4961.9 1865.78  4995.1 1866.96  5002.2 1866.39  5016.5 1863.34    5017 1862.84
  5028.5 1863.34  5083.5 1869.71  5124.1 1869.57  5162.5 1871.93  5266.4 1873.84
  5280.2 1874.83  5347.6  1875.1  5571.1 1879.07    6015 1884.65  6375.5  1888.2
#Mann= 6 ,-1 , 0
  3831.6     .12       0  3992.1     .05       0  4192.4     .12       0
  4292.6     .05       0  5016.5     .05       0  5028.5     .05       0
Bank Sta=5016.5,5028.5
XS Rating Curve= 0 ,0
Exp/Cntr=0.3,0.1

Type RM Length L Ch R = 1 ,24647   ,519,519,519
BEGIN DESCRIPTION:
Elm 01 91 24647.25
END DESCRIPTION:
XS GIS Cut Line= 3
       1604055.9      6797033.19      1605310.26      6796833.54
      1606290.57      6796590.63
#Sta/Elev= 30
  3731.7 1896.26  3753.4 1895.46    3832 1893.27  3913.1 1890.18  3948.3 1888.11
  4166.2 1880.89  4186.4 1879.37    4242 1878.95  4304.2 1876.69  4371.4 1875.88
  4620.2 1870.18  4682.4 1869.97    4794 1866.34  4976.3 1864.89  5001.9 1861.58
  5002.4 1861.08  5014.1 1861.58  5027.3 1865.64  5078.8 1865.04  5109.8 1863.06
    5127  1864.8  5132.2 1866.67  5161.3 1868.65  5173.5 1870.57  5202.5 1872.71
  5274.6 1873.59  5346.7 1875.82  5421.9 1876.06  5470.3 1877.48  6011.8 1884.79
#Mann= 5 ,-1 , 0
  3731.7     .05       0  3753.4     .12       0  3948.3     .05       0
  5001.9     .05       0  5014.1     .05       0
Bank Sta=5001.9,5014.1
XS Rating Curve= 0 ,0
Exp/Cntr=0.3,0.1

Type RM Length L Ch R = 1 ,24128   ,180,180,180
BEGIN DESCRIPTION:
Elm 01 91 24128.18
END DESCRIPTION:
XS GIS Cut Line= 5
      1604512.47      6797100.72      1605410.08      6797081.63
      1605538.56      6797038.22       1605713.9       6797046.9
      1606297.21      6796954.89
#Sta/Elev= 30
  3791.9 1879.97  4124.5 1871.73  4444.6 1867.88  4574.6  1867.5  4584.6 1867.08
  4614.6 1861.28    4636 1861.85  4654.6 1862.71  4674.6 1866.04  4713.7 1869.02
  4795.8 1870.07  4831.8 1870.49  4861.8 1862.26  4871.8 1861.75  4924.4 1862.49
  4976.4 1861.58    4992 1860.87  4992.8 1859.36  4993.3 1858.86  5005.1 1859.36
  5021.6 1860.19  5032.4 1863.82  5062.7 1868.64  5089.1  1874.7  5133.6 1875.72
  5174.1 1874.79    5222 1877.14  5265.2 1876.73  5396.8 1880.74  5591.4  1883.1
#Mann= 7 ,-1 , 0
  3791.9     .05       0    4636     .12       0  4795.8     .05       0
  4976.4     .12       0  4992.8     .07       0  5005.1     .12       0
    5222     .05       0
Bank Sta=4992.8,5005.1
XS Rating Curve= 0 ,0
Exp/Cntr=0.3,0.1

Type RM Length L Ch R = 1 ,23948   ,466,466,466
BEGIN DESCRIPTION:
Elm 01 91 23947.9
END DESCRIPTION:
XS GIS Cut Line= 3
      1604734.77      6797213.57      1605807.65        6797191.
       1606361.6      6797178.88
#Sta/Elev= 30
  3929.6 1877.66  3960.8 1877.24  3979.8  1873.8  4019.8 1871.46  4049.9 1871.66
  4084.5 1870.61  4099.9 1870.96  4159.9 1869.26    4590 1866.32    4650 1865.02
    4740 1861.73    4790 1861.12    4890  1860.6  4990.1 1861.47  5010.1 1860.47
  5023.9  1858.9  5024.4  1858.4  5035.7  1858.4  5036.2  1858.9  5040.1 1860.69
  5050.1 1862.55  5160.1 1863.44  5220.1 1865.16  5240.1 1866.53  5273.1 1871.71
  5290.1 1874.44  5336.6  1877.6  5360.2 1877.83  5371.8  1878.9  5556.8 1881.87
#Mann= 6 ,-1 , 0
  3929.6     .12       0  4084.5     .05       0  5023.9     .05       0
  5036.2     .05       0  5273.1     .12       0  5336.6     .05       0
Bank Sta=5023.9,5036.2
XS Rating Curve= 0 ,0
Exp/Cntr=0.3,0.1

Type RM Length L Ch R = 1 ,23482   ,521,521,521
BEGIN DESCRIPTION:
Elm 01 91 23797.67
END DESCRIPTION:
XS GIS Cut Line= 3
      1604923.95      6797335.09      1605760.03      6797542.84
      1606580.31       6797303.1
#Sta/Elev= 30
  4138.5 1874.49  4140.7 1874.49  4149.9 1874.75  4168.3 1871.45  4221.9 1869.51
  4726.9 1864.86  4943.3 1857.22  4984.5 1858.44  5005.2 1857.82  5015.6 1859.99
  5066.6  1858.7  5071.8  1857.2  5098.9 1858.93  5138.7 1858.57  5143.9 1856.34
  5152.7 1855.41  5153.2 1854.91  5170.3 1855.41  5213.4  1857.5  5234.4 1857.88
  5255.2 1856.58  5276.1  1858.8    5455 1860.34  5566.2 1863.26  5578.2 1865.26
    5610 1867.42  5638.3 1867.55  5710.4 1873.68  5765.7 1880.84  5854.6 1883.61
#Mann= 7 ,-1 , 0
  4138.5     .05       0  4140.7     .12       0  4221.9     .05       0
  5152.7     .03       0  5170.3     .05       0  5213.4     .12       0
    5455     .05       0
Bank Sta=5152.7,5170.3
XS Rating Curve= 0 ,0
Exp/Cntr=0.3,0.1

Type RM Length L Ch R = 1 ,22961   ,963,963,963
BEGIN DESCRIPTION:
Elm 01 91 22961.21
END DESCRIPTION:
XS GIS Cut Line= 4
      1605814.27      6798483.51       1605957.5      6797776.01
      1606230.94      6797567.68       1606586.6      6797402.87
#Sta/Elev= 30
  3932.1 1864.03  4141.8 1861.91  4382.5 1861.63  4519.9 1861.53  4549.9 1862.28
  4611.1 1861.03  4616.2 1861.59  4664.3  1858.9  4701.1 1858.08  4883.3  1858.2
  4957.4  1857.9  4971.9 1856.92  4986.4 1857.03  4992.7 1855.81  5008.3  1855.9
  5015.4 1855.13  5015.9 1854.63  5032.5 1854.63    5033 1855.13  5036.7 1859.39
  5122.8 1860.14  5145.5 1861.48  5151.3 1862.61  5174.2 1863.15  5233.6 1869.28
  5248.4 1872.14  5255.7  1874.6  5277.7 1878.56  5317.2 1880.71  5389.7  1882.8
#Mann= 5 ,-1 , 0
  3932.1     .05       0  4382.5     .12       0  4883.3     .05       0
  5015.4     .05       0    5033     .05       0
Bank Sta=5015.4,5033
XS Rating Curve= 0 ,0
Exp/Cntr=0.3,0.1

Type RM Length L Ch R = 1 ,21998   ,643,643,643
BEGIN DESCRIPTION:
Elm 01 91 21997.54
END DESCRIPTION:
XS GIS Cut Line= 3
      1605866.35      6798943.56      1606200.56      6798188.34
      1606638.95      6797524.25
#Sta/Elev= 30
  4172.8 1872.46  4244.5 1870.83    4253 1870.31  4258.4 1868.39  4288.2 1866.32
  4342.9 1864.16  4374.9 1864.23  4409.1 1862.82  4554.3 1860.07  4747.1 1859.26
  4769.4 1859.83  4813.1 1858.22  4920.1 1856.66  4966.2 1857.16  4977.6 1855.83
  4986.6 1850.88  4987.1 1850.38  5004.3 1850.88  5010.4 1853.33  5046.6 1854.76
  5154.8 1855.14    5355 1858.88  5609.5 1864.55  5651.6 1867.01  5687.7 1870.49
  5717.9 1874.88  5723.9 1875.02  5738.9 1878.44    5760    1880  5794.4 1880.78
#Mann= 5 ,-1 , 0
  4172.8     .05       0  4747.1     .12       0  4986.6     .07       0
  5004.3     .12       0    5355     .05       0
Bank Sta=4986.6,5004.3
XS Rating Curve= 0 ,0
Exp/Cntr=0.3,0.1

Type RM Length L Ch R = 1 ,21355   ,629,629,629
BEGIN DESCRIPTION:
Elm 01 91 21354.76
END DESCRIPTION:
XS GIS Cut Line= 3
      1605970.55      6799056.37      1606586.85       6798561.6
      1607946.28      6797699.26
#Sta/Elev= 30
  4214.6 1873.51  4245.7 1872.96    4273 1869.61  4309.7  1868.1  4359.4 1863.46
  4423.4 1861.11  4586.6 1858.15  4813.8  1855.9  4842.6 1854.49  4941.8 1852.69
  4999.4 1854.23  5014.6 1851.37  5017.8 1847.69  5018.3 1847.19  5035.6 1847.69
  5057.2 1853.41  5114.8 1853.63  5208.8 1856.33  5296.9 1856.14  5339.3 1857.29
  5500.1 1856.73  5636.7 1858.01  5673.1 1859.44  5818.8 1860.35  6106.9 1866.51
  6252.6 1867.12  6310.2 1869.43  6340.7 1867.86  6519.5 1871.13  6614.8 1871.07
#Mann= 3 ,-1 , 0
  4214.6     .05       0  5017.8     .05       0  5035.6     .05       0
Bank Sta=5017.8,5035.6
XS Rating Curve= 0 ,0
Exp/Cntr=0.3,0.1

Type RM Length L Ch R = 1 ,20726   ,1447,1447,1447
BEGIN DESCRIPTION:
Elm 01 91 20725.67
END DESCRIPTION:
XS GIS Cut Line= 3
      1606044.35      6799052.05      1606855.94      6798999.97
      1608400.51      6798947.91
#Sta/Elev= 30
    4186 1868.85  4236.8 1864.65  4296.9 1862.06  4324.6 1861.79    4337 1860.66
  4617.5 1856.31  4667.6 1856.29  4878.1 1852.36  5001.3 1851.81  5008.3 1850.16
  5009.3 1847.55  5009.8 1847.05  5027.4 1847.55  5028.3 1851.04  5038.3 1851.63
  5218.4 1852.07  5248.5 1852.85  5285.2  1851.7  5378.5 1849.79  5398.5 1847.92
  5412.6 1848.38  5428.6 1850.42  5478.6 1849.48  5508.6 1850.99  5708.7 1857.26
  5768.8 1860.31  5868.8 1862.51  6001.3 1863.93  6309.1 1868.56  6544.7 1873.39
#Mann= 6 ,-1 , 0
    4186     .05       0  5009.3     .05       0  5027.4     .05       0
  5285.2     .12       0  5412.6     .05       0  6001.3     .12       0
Bank Sta=5009.3,5027.4
XS Rating Curve= 0 ,0
Exp/Cntr=0.3,0.1

Type RM Length L Ch R = 1 ,19279   ,193,193,193
BEGIN DESCRIPTION:
Mapping XS d450de37
END DESCRIPTION:
XS GIS Cut Line= 5
      1606204.06      6799477.42      1607224.88      6799532.98
      1607353.85      6799457.49      1607804.37      6799309.06
      1608408.09      6799133.28
#Sta/Elev= 30
  3563.6 1870.27  3644.7 1860.41  3684.7 1857.65  3724.8 1856.41  4475.9 1849.56
    4576 1854.85  4604.6 1855.19  4620.3 1854.61  4647.5 1851.37  4663.2 1852.79
  4684.7 1853.08  4757.6 1850.14  4799.8 1850.52  4809.3 1848.99  4814.6 1842.61
  4820.8 1839.05  4831.3 1836.26  4927.3 1835.26  4927.8 1834.76  4945.5 1835.26
  4999.8 1836.29  5005.2 1840.12  5010.5 1840.59  5020.9 1846.32  5031.4 1849.02
  5169.3 1851.67  5339.6 1857.02    5502 1863.91  5551.1 1867.45  5838.5 1872.42
#Mann= 3 ,-1 , 0
  3563.6     .05       0  4927.3     .05       0  4945.5     .05       0
Bank Sta=4927.3,4945.5
XS Rating Curve= 0 ,0
Exp/Cntr=0.3,0.1

Type RM Length L Ch R = 1 ,19086   ,60,60,60
BEGIN DESCRIPTION:
Mapping XS 9cf1aa75
END DESCRIPTION:
XS GIS Cut Line= 4
      1606464.49      6799612.84       1607437.3      6799573.71
      1608155.61      6799547.66      1608416.04      6799521.62
#Sta/Elev= 30
    3859 1859.48  3919.6 1855.97  4029.6 1853.85    4500 1849.25  4598.2  1849.9
  4720.2 1855.39  4740.2 1855.96  4770.2  1855.6  4848.7 1850.44  4890.3 1849.17
  4900.3 1846.89  4910.3 1841.31  4920.3 1836.92  4930.4 1835.69  4961.3 1835.23
  4961.8 1834.73    4979 1834.73  4979.5 1835.23  5000.4 1835.45  5010.4 1838.57
  5030.4 1849.79  5050.4  1849.3  5160.5 1849.54  5380.7 1854.04  5450.7 1858.37
  5490.7 1864.16  5548.6 1868.21  5721.6 1873.56  5751.8 1873.88  5813.1  1872.7
#Mann= 3 ,-1 , 0
    3859     .05       0  4961.3     .05       0  4979.5     .05       0
Bank Sta=4961.3,4979.5
XS Rating Curve= 0 ,0
Exp/Cntr=0.3,0.1

Type RM Length L Ch R = 1 ,19026   ,195,195,195
BEGIN DESCRIPTION:
Mapping XS c76bd12b
END DESCRIPTION:
XS GIS Cut Line= 3
      1606481.82      6799682.28       1607524.1       6799632.3
      1608320.25      6799591.08
#Sta/Elev= 30
  3876.1 1859.12  3919.3 1856.21  4067.2 1853.42  4419.9 1849.58  4570.1 1849.85
  4580.1 1848.72  4610.1 1840.89  4620.1 1839.09  4630.1 1838.83  4660.2 1839.81
  4690.2 1842.29  4740.3 1854.11  4750.3 1855.86  4760.3 1856.29  4800.3 1854.92
  4890.4 1848.41  4970.5 1845.81  4980.6  1843.9  4990.6 1840.32  4991.5 1838.17
    4992 1837.67  5009.7 1838.17  5010.6 1842.14  5020.6  1847.4  5030.6  1848.7
  5190.8 1849.23  5381.1 1853.29  5451.2 1857.42  5486.3 1862.98  5716.8 1873.12
#Mann= 3 ,-1 , 0
  3876.1     .05       0  4991.5     .05       0  5009.7     .05       0
Bank Sta=4991.5,5009.7
XS Rating Curve= 0 ,0
Exp/Cntr=0.3,0.1

Type RM Length L Ch R = 1 ,18831   ,420,420,420
BEGIN DESCRIPTION:
Mapping XS 2e266f0a
END DESCRIPTION:
XS GIS Cut Line= 3
      1606401.92      6799782.97      1607448.15       6799821.1
      1608055.79      6799827.61
#Sta/Elev= 30
  3797.4 1860.76  3860.5 1853.71  3900.6 1852.65  4490.9 1849.31  4500.9 1848.92
    4511 1846.74  4551.9 1835.41  4552.4 1834.91  4570.1 1835.41    4624 1835.41
  4681.1 1850.59  4691.1 1852.56  4721.1 1855.34  4771.1 1854.04  4821.2 1849.89
  4881.2 1847.16  4951.2  1845.9  4961.2 1839.93  4971.2 1835.41  4981.2 1835.41
  4991.2 1836.54  5001.2 1844.36  5011.2 1847.19  5101.2 1848.07  5261.2 1847.98
  5341.2 1849.06  5401.2 1850.51  5421.2 1852.66  5441.2 1856.72    5452  1856.8
#Mann= 3 ,-1 , 0
  3797.4     .05       0  4551.9     .04       0  4570.1     .05       0
Bank Sta=4551.9,4570.1
XS Rating Curve= 0 ,0
Exp/Cntr=0.3,0.1

Type RM Length L Ch R = 1 ,18411   ,226,226,226
BEGIN DESCRIPTION:
Mapping XS b3091b88
END DESCRIPTION:
XS GIS Cut Line= 4
      1606614.83      6800042.46       1606899.1      6800135.77
      1607979.83      6800196.54      1608539.68      6800094.55
#Sta/Elev= 30
  4194.6 1850.49  4436.9 1849.16  4579.8 1847.71  4639.9 1846.38  4790.2  1846.6
  4810.2 1846.15  4840.2  1846.6  4930.4    1846  4950.4 1844.78  4960.4 1840.92
  4961.3  1835.4  4961.8  1834.9    4979  1834.9  4979.5  1835.4  4982.2  1837.7
  5000.5 1841.87  5010.5 1844.82  5020.5 1846.34  5110.7 1845.81  5210.8  1846.1
  5421.2 1843.89  5514.8 1843.72  5642.5 1845.63  5662.8 1847.26    5703 1847.12
  5886.4  1851.6  6069.4 1853.88  6101.5 1855.33    6110 1854.72  6145.3 1854.98
#Mann= 3 ,-1 , 0
  4194.6     .05       0  4961.3     .06       0  4979.5     .05       0
Bank Sta=4961.3,4979.5
XS Rating Curve= 0 ,0
Exp/Cntr=0.3,0.1

Type RM Length L Ch R = 1 ,18185   ,1068,1068,1068
BEGIN DESCRIPTION:
Elm 01 91 18185.38
END DESCRIPTION:
XS GIS Cut Line= 3
      1606398.14      6800364.27      1607405.13      6800390.31
      1608271.63      6800411.97
#Sta/Elev= 30
  3993.3    1847  4060.2 1846.47  4140.2 1846.84  4390.3 1844.64  4640.4 1844.93
  4870.5 1844.26  4890.5  1844.3  4930.5 1845.67  4940.5 1845.57  4950.5 1845.29
  4960.5 1843.54  4970.5  1837.9    4989 1833.51  4989.5 1833.01  5006.7 1833.01
  5007.2 1833.51  5010.5 1834.71  5020.5 1841.69  5030.5  1844.2  5160.5 1844.03
  5230.6 1844.81  5360.6 1844.02  5420.6 1844.12  5520.7 1842.99  5570.7 1842.96
  5630.7 1843.85  5640.7 1843.65  5660.7 1845.03  5710.7 1844.78  5867.4  1846.5
#Mann= 3 ,-1 , 0
  3993.3     .05       0    4989     .04       0  5007.2     .05       0
Bank Sta=4989,5007.2
XS Rating Curve= 0 ,0
Exp/Cntr=0.3,0.1

Type RM Length L Ch R = 1 ,17117   ,696,696,696
BEGIN DESCRIPTION:
Elm 01 91 17117.38
END DESCRIPTION:
XS GIS Cut Line= 3
      1606730.04      6800966.14      1608209.82      6800965.31
      1608810.24      6800965.31
#Sta/Elev= 30
  3524.8 1844.83  3649.8 1843.88  3689.8 1842.54  3719.8  1843.1  3739.8 1841.92
  3829.8 1840.29  4149.8 1841.76  4379.8  1841.3  4449.8 1840.41  4489.8 1841.77
  4609.8 1840.58  4679.8 1841.57  4859.8 1841.49  4969.8 1839.43  4979.8 1836.16
  4980.6 1833.67  4981.1 1833.17  4998.9 1833.67  4999.7 1836.18  5004.6 1836.18
  5009.8 1840.77  5019.8 1843.25  5029.8 1844.67  5059.8 1844.02  5229.8 1843.95
  5329.8  1845.6  5339.8 1846.51  5409.8 1845.96  5469.8  1847.2    5605 1847.65
#Mann= 3 ,-1 , 0
  3524.8     .05       0  4980.6     .05       0  4998.9     .05       0
Bank Sta=4980.6,4998.9
XS Rating Curve= 0 ,0
Exp/Cntr=0.3,0.1

Type RM Length L Ch R = 1 ,16421   ,1119,1119,1119
BEGIN DESCRIPTION:
Elm 01 91 16420.72
END DESCRIPTION:
XS GIS Cut Line= 3
       1606918.1       6801479.2      1607758.43      6801430.59
      1608654.28      6801381.97
#Sta/Elev= 30
  4160.1 1841.83  4387.4  1840.4  4397.4 1840.63  4417.4 1842.69  4427.4  1841.1
  4447.5 1840.35  4627.8 1839.85  4838.1  1837.3  4978.4 1839.92  5001.8 1838.04
  5008.4 1836.08  5009.3 1834.63  5009.8 1834.13  5027.6 1834.63  5028.4 1836.37
  5038.5 1837.05  5088.5  1837.6  5108.6 1836.92  5142.7 1839.56  5188.7 1838.76
  5258.8 1838.88  5368.9 1841.55    5419 1841.54  5469.1 1843.09  5619.3 1845.01
  5669.4 1846.56  5769.5 1846.35  5789.6 1847.48  5829.6    1846    5899 1845.47
#Mann= 3 ,-1 , 0
  4160.1     .05       0  5009.3     .05       0  5027.6     .05       0
Bank Sta=5009.3,5027.6
XS Rating Curve= 0 ,0
Exp/Cntr=0.3,0.1

Type RM Length L Ch R = 1 ,15302   ,607,607,607
BEGIN DESCRIPTION:
Elm 01 91 15302.18
END DESCRIPTION:
XS GIS Cut Line= 3
      1607172.34      6801996.79      1608307.74      6801989.85
      1608838.97       6801982.9
#Sta/Elev= 30
  3863.5 1838.84  3946.2 1839.25  3996.2 1838.09  4196.2 1837.08  4266.2 1837.59
  4396.2 1835.16  4536.2 1835.25  4586.2 1833.68  4610.7 1835.59  4776.2 1837.24
  4806.2 1836.56  4836.2 1831.28  4846.2 1831.96  4856.2  1836.2  4886.2 1835.36
  4966.2  1836.9  4986.2 1836.08  4995.1 1832.27    4997 1830.22  4997.5 1829.72
  5015.3 1830.22  5016.2 1832.28  5026.2 1834.75  5046.2 1834.88  5066.2 1833.76
  5096.2 1834.45  5136.2 1837.13  5151.9 1836.95  5236.2 1836.92  5530.2 1839.59
#Mann= 5 ,-1 , 0
  3863.5     .05       0  4610.7     .12       0    4997     .07       0
  5015.3     .12       0  5151.9     .05       0
Bank Sta=4997,5015.3
XS Rating Curve= 0 ,0
Exp/Cntr=0.3,0.1

Type RM Length L Ch R = 1 ,14695   ,540,540,540
BEGIN DESCRIPTION:
Elm 01 91 14694.5
END DESCRIPTION:
XS GIS Cut Line= 3
      1607182.76       6802382.2      1608050.79      6802288.46
      1608877.19      6802253.73
#Sta/Elev= 30
  4130.6 1837.81  4173.1 1837.36  4223.4    1838  4309.2 1836.39    4401 1836.26
  4484.9 1835.11  4665.9 1835.85  4796.7 1834.98  4865.2 1833.44  4877.2 1833.83
  4887.2 1835.23  4907.3 1834.57  4927.4 1832.79  4967.7 1832.23  4978.4 1828.93
  4978.9 1828.43  4996.6 1828.43  4997.1 1828.93  4997.9 1831.91  5008.3 1831.59
  5017.9 1833.29  5067.9 1835.58    5108 1833.38    5158 1832.18  5218.1 1834.27
  5298.1 1833.31  5408.2 1833.08  5448.3 1834.78  5498.3 1833.96  5830.8  1837.6
#Mann= 3 ,-1 , 0
  4130.6     .05       0  4978.4     .05       0  4997.1     .05       0
Bank Sta=4978.4,4997.1
XS Rating Curve= 0 ,0
Exp/Cntr=0.3,0.1

Type RM Length L Ch R = 1 ,14155   ,621,621,621
BEGIN DESCRIPTION:
Elm 01 91 14154.67
END DESCRIPTION:
XS GIS Cut Line= 3
       1607144.5      6802705.12      1607870.24      6802719.01
      1608908.38      6802507.22
#Sta/Elev= 30
  4268.6 1836.74  4449.1 1836.43  4509.1 1835.45  4779.2 1833.83  4789.2 1834.43
  4839.2  1832.7  4899.2 1834.17  4949.2 1834.14  4969.2  1830.3  4969.9 1827.67
  4970.4 1827.17  4988.1 1827.17  4988.6 1827.67  4989.2 1828.48  4994.3 1830.04
  5019.6 1831.45  5029.9  1830.4  5070.1 1833.48  5075.2 1832.99    5081 1833.71
  5101.4    1834  5170.9 1833.92  5193.2 1833.89  5221.7 1832.33  5285.1 1833.34
  5356.5 1833.44  5540.2 1831.25  5632.1  1831.9  5662.7 1830.99    6054 1835.43
#Mann= 4 ,-1 , 0
  4268.6     .05       0  4969.9     .07       0  4988.6     .05       0
  5170.9     .05       0
Bank Sta=4969.9,4988.6
XS Rating Curve= 0 ,0
Exp/Cntr=0.3,0.1

Type RM Length L Ch R = 1 ,13534   ,469,469,469
BEGIN DESCRIPTION:
Elm 01 91 13534.47
END DESCRIPTION:
XS GIS Cut Line= 4
      1607264.74      6803370.93      1607957.04      6803177.78
      1608504.78      6802892.06      1609020.51      6802587.64
#Sta/Elev= 30
    4283 1835.45    4345 1834.27  4698.5 1833.72  4854.3 1831.43    4949 1831.55
  4958.1 1831.35    4978  1827.9  4979.6 1827.05  4980.1 1826.55  4998.3 1826.55
  4998.8 1827.05  5001.7 1830.12  5008.6 1831.53    5022 1832.42  5058.4 1831.94
  5074.8 1830.63  5080.5 1829.38  5096.9 1828.34  5102.6 1829.68  5124.7 1830.58
  5201.7 1830.71    5304  1832.7  5483.3  1831.5  5615.8 1831.99  5666.2 1830.61
  5791.4 1829.93  6111.4 1833.71  6191.4 1833.73    6207 1835.33  6218.4 1835.33
#Mann= 3 ,-1 , 0
    4283     .05       0  4979.6     .05       0  4998.8     .05       0
Bank Sta=4979.6,4998.8
XS Rating Curve= 0 ,0
Exp/Cntr=0.3,0.1

Type RM Length L Ch R = 1 ,13065   ,1024,1024,1024
BEGIN DESCRIPTION:
Mapping XS 0d9294b1
END DESCRIPTION:
XS GIS Cut Line= 5
      1607340.96      6803848.86      1607853.96       6803489.5
      1608054.48      6803335.86      1608421.67      6803044.19
      1608993.03      6802642.02
#Sta/Elev= 30
  4443.9  1832.5  4856.4 1832.45  4913.1 1830.47  4927.9 1828.36  4942.7  1825.2
  4947.9 1823.38  4948.4 1822.88  4967.1 1823.38  4999.4 1824.73  5008.1 1825.76
  5014.2 1827.74    5029 1830.42  5043.9 1830.81  5108.4 1830.23  5185.4 1831.59
  5325.2 1830.85  5392.8 1829.31  5456.8  1829.4  5477.7 1827.51  5485.7 1829.19
  5492.1 1829.48  5613.9 1831.24  5677.9 1830.97  5748.4  1831.9  5820.3    1831
    5878 1832.36  5913.8 1830.69  6121.9  1829.9  6466.9 1833.24  6490.5 1834.84
#Mann= 3 ,-1 , 0
  4443.9     .05       0  4947.9     .05       0  4967.1     .05       0
Bank Sta=4947.9,4967.1
XS Rating Curve= 0 ,0
Exp/Cntr=0.3,0.1

Type RM Length L Ch R = 1 ,12041   ,467,467,467
BEGIN DESCRIPTION:
Mapping XS 800fa10a
END DESCRIPTION:
XS GIS Cut Line= 5
      1607679.51       6803999.9        1608380.      6803523.36
      1608643.02      6803197.84       1608692.5      6802960.86
      1608974.41      6802683.62
#Sta/Elev= 30
  3860.6 1831.33  4405.8 1830.41  4420.8 1829.77  4471.6  1829.9  4520.3 1828.15
  4585.4 1827.44  4693.2 1829.54  4707.8 1828.93  4722.4 1829.47    4772 1828.77
  4864.7 1828.91  4935.1 1827.52  4963.9 1827.09  4984.7 1824.59  4992.7  1824.9
  5003.9 1824.05  5004.4 1823.55  5022.6 1823.55  5023.1 1824.05  5027.9 1828.25
  5035.8 1828.19    5049 1829.57  5188.8 1830.04  5269.2 1830.79  5311.2 1829.36
  5400.4 1829.57  5718.7  1832.5  5732.9  1833.4    5754 1833.33  5763.8 1834.25
#Mann= 5 ,-1 , 0
  3860.6     .05       0  4935.1     .12       0  5003.9     .07       0
  5023.1     .12       0  5188.8     .05       0
Bank Sta=5003.9,5023.1
XS Rating Curve= 0 ,0
Exp/Cntr=0.3,0.1

Type RM Length L Ch R = 1 ,11574   ,403,403,403
BEGIN DESCRIPTION:
Elm 01 91 11573.622
END DESCRIPTION:
XS GIS Cut Line= 3
      1607604.82      6804112.08        1608803.      6803643.37
      1609536.92      6803170.25
#Sta/Elev= 30
  3713.4 1830.77  3724.3 1830.44  3739.4 1831.15  3756.5 1829.87  3793.7 1831.32
  4065.2 1829.93  4287.7 1830.17  4504.9 1828.14    4680 1827.72  4697.6 1826.66
  4765.9 1825.85  4819.6 1825.84  4873.3 1827.18  4920.1 1826.75    4950 1825.28
  4987.8 1822.17  4988.3 1821.67  5008.9 1822.17  5019.7 1824.95  5026.2 1825.15
  5085.7 1825.21  5092.3 1825.99  5113.4 1825.25  5149.7 1826.67  5160.4 1826.36
  5367.5 1828.16  5373.5 1829.05    5555 1829.61  5656.8 1831.68  5873.2 1833.71
#Mann= 4 ,-1 , 0
  3713.4     .05       0  4987.8     .05       0  5008.9     .05       0
  5160.4     .05       0
Bank Sta=4987.8,5008.9
XS Rating Curve= 0 ,0
Exp/Cntr=0.3,0.1

Type RM Length L Ch R = 1 ,11171   ,613,613,613
BEGIN DESCRIPTION:
Elm 01 91 11170.66
END DESCRIPTION:
XS GIS Cut Line= 3
      1607678.52      6804229.29      1608728.92      6804012.27
      1609705.52      6803400.27
#Sta/Elev= 30
  3928.5 1830.74  4060.6 1829.64  4088.3  1828.3  4118.9 1829.37  4486.5 1828.23
    4603 1828.44  4629.5 1830.21  4703.5 1830.81  4748.6 1828.71  4833.7 1829.15
  4884.8 1828.35  4935.8 1825.78  4976.7 1821.83  4986.9  1822.1  4988.7 1820.62
  4989.2 1820.12  5009.8 1820.62  5016.3 1822.24  5043.7 1822.35  5052.9 1823.48
    5080 1824.79  5089.4 1824.41  5116.5 1826.48  5168.4 1825.72  5283.1 1826.46
  5320.4 1826.56  5335.7 1825.09  5350.5 1825.05  5633.7  1826.2  6153.6 1832.72
#Mann= 4 ,-1 , 0
  3928.5     .05       0  4988.7     .05       0  5009.8     .12       0
  5283.1     .05       0
Bank Sta=4988.7,5009.8
XS Rating Curve= 0 ,0
Exp/Cntr=0.3,0.1

Type RM Length L Ch R = 1 ,10558   ,251,251,251
BEGIN DESCRIPTION:
Elm 01 91 10557.84
END DESCRIPTION:
XS GIS Cut Line= 3
      1607356.53      6804332.58      1609169.02      6804297.86
      1611054.47      6804287.44
#Sta/Elev= 30
  3188.8 1830.26  3477.3 1830.23  3717.4 1827.91  4177.5 1827.23  4197.5 1828.47
  4227.5 1827.31  4757.6 1824.76  4847.6 1825.41  4947.6 1822.56  4977.6 1818.71
  4987.6  1820.6  5037.6 1818.43  5077.6 1822.25  5087.1 1817.36  5087.6 1816.86
  5108.2 1817.36  5117.6 1822.64  5157.6 1825.88  5177.6 1824.14  5447.6 1823.37
  5477.6 1830.71  5487.6 1831.12  5527.6 1824.72  5547.6 1819.39  5557.6 1819.36
  5617.6  1819.4  5647.6 1824.23  5667.6 1823.01  6197.6 1824.82  6887.1 1829.56
#Mann= 3 ,-1 , 0
  3188.8     .05       0  5087.1     .03       0  5108.2     .05       0
Bank Sta=5087.1,5108.2
XS Rating Curve= 0 ,0
Exp/Cntr=0.3,0.1

Type RM Length L Ch R = 1 ,10307   ,580,580,580
BEGIN DESCRIPTION:
Elm 01 91 10306.82
END DESCRIPTION:
XS GIS Cut Line= 3
      1607618.51       6804577.7      1609254.78      6804521.28
      1610851.02      6804495.25
#Sta/Elev= 30
    3361 1828.09  3587.6 1826.66  3767.7 1827.16  3907.8 1826.18    4228 1826.19
    4268 1826.89  4358.1  1825.2  4418.1 1825.63  4698.3 1823.91  4828.4 1825.17
  4945.8 1820.59  4977.8 1816.81  4978.3 1816.31  4998.6 1816.31  4999.1 1816.81
  5000.9  1817.8  5008.5 1819.52  5038.5 1821.99  5108.5 1823.12  5118.5 1823.86
  5458.5 1822.45  5588.5  1820.6  5938.6 1822.52  6038.6 1824.04  6108.6 1826.71
  6158.6 1827.26  6438.7  1828.2  6458.7 1828.95  6538.7 1828.26  6594.7 1828.58
#Mann= 3 ,-1 , 0
    3361     .05       0  4977.8     .05       0  4999.1     .05       0
Bank Sta=4977.8,4999.1
XS Rating Curve= 0 ,0
Exp/Cntr=0.3,0.1

Type RM Length L Ch R = 1 ,9727    ,536,536,536
BEGIN DESCRIPTION:
Elm 01 91 9727.4
END DESCRIPTION:
XS GIS Cut Line= 4
      1608518.72      6805060.26      1608869.59      6805070.98
      1609723.53      6804807.73      1610660.47      6804651.58
#Sta/Elev= 30
  3754.4 1824.81  3790.7 1823.15  3850.7 1822.98  3860.7  1823.5  3920.8 1822.26
  4080.8  1821.9  4841.9 1822.76  4879.8 1821.91  4945.1 1821.83    4983 1819.43
    5000 1816.06  5000.5 1815.56  5020.8 1815.56  5021.3 1816.06  5026.8 1818.68
  5031.9 1819.71  5041.1 1818.62  5061.4 1820.26  5148.5 1821.86  5162.7 1821.33
    5254 1821.98  5275.2 1820.03  5324.9 1819.06  5391.8  1820.3    5477 1820.44
  5518.5 1821.73  5568.2 1821.91  5649.4 1823.72    5696 1823.39  5948.9 1827.09
#Mann= 3 ,-1 , 0
  3754.4     .05       0    5000     .05       0  5021.3     .05       0
Bank Sta=5000,5021.3
XS Rating Curve= 0 ,0
Exp/Cntr=0.3,0.1

Type RM Length L Ch R = 1 ,9191    ,1011,1011,1011
BEGIN DESCRIPTION:
Mapping XS fca7e6ed
END DESCRIPTION:
XS GIS Cut Line= 6
      1608516.54      6805181.79      1609572.67      6805228.44
      1609925.68      6805191.54      1610268.57      6804952.83
      1610361.88      6804790.07      1610670.03      6804696.76
#Sta/Elev= 30
  3405.4 1824.47  3430.9 1822.86  3674.1 1821.31  4084.5 1822.48  4404.8 1820.51
  4926.3 1821.65  4976.8 1819.17  4991.7 1815.85  4995.8 1812.81  4996.3 1812.31
  5017.2 1812.81  5021.3 1817.36  5042.3 1820.92  5128.7 1820.67  5143.5 1821.21
  5149.6 1823.81  5164.5 1822.14  5194.1 1823.34  5200.2 1821.62  5215.1 1823.42
  5235.1 1822.74  5257.9 1824.37  5273.4 1823.32  5300.5 1825.31  5354.2 1823.68
  5359.9 1821.85  5403.3 1820.25  5645.6 1825.31  5697.9 1825.14  5744.9 1827.13
#Mann= 3 ,-1 , 0
  3405.4     .05       0  4995.8     .05       0  5017.2     .05       0
Bank Sta=4995.8,5017.2
XS Rating Curve= 0 ,0
Exp/Cntr=0.3,0.1

Type RM Length L Ch R = 1 ,8180    ,338,338,338
BEGIN DESCRIPTION:
Mapping XS c83c849c
END DESCRIPTION:
XS GIS Cut Line= 5
      1608518.78      6805220.85      1609481.65      6805276.04
      1610279.42      6805302.22      1610531.15      6805221.93
      1610980.21      6804968.11
#Sta/Elev= 30
    2857 1824.15  2883.3 1822.87  3103.6 1821.08    3414 1821.44  3674.6 1820.35
  4345.1  1821.1  4415.1 1817.41  4435.1 1818.02  4455.1 1821.08  4485.2 1820.08
  4575.2 1820.45  4645.6 1819.49  4844.1 1818.31  4849.3  1818.8  4883.9 1817.96
  4925.4 1818.31  4957.2 1816.75  4968.2 1813.91  4968.7 1813.41  4989.1 1813.41
  4989.6 1813.91  4991.7 1816.95  5006.3 1820.43  5029.3 1822.39  5043.8 1821.99
  5048.6  1822.5  5124.7 1822.21  5264.7 1825.59  5329.7 1825.32  5399.7 1827.11
#Mann= 5 ,-1 , 0
    2857     .05       0  4968.2     .05       0  4989.6     .05       0
  5029.3     .12       0  5048.6     .05       0
Bank Sta=4968.2,4989.6
XS Rating Curve= 0 ,0
Exp/Cntr=0.3,0.1

Type RM Length L Ch R = 1 ,7842    ,229,229,229
BEGIN DESCRIPTION:
Mapping XS d580d016
END DESCRIPTION:
XS GIS Cut Line= 5
      1608518.73      6805246.89      1609321.09      6805293.29
      1610431.33      6805339.11      1610646.17      6805538.77
      1610917.39      6805601.69
#Sta/Elev= 30
  3013.4 1823.67  3039.7 1822.57  3149.9  1822.2    3240 1820.91  3330.2 1822.23
  3400.3 1820.76  3642.3 1820.76  3670.8 1821.36  3814.1 1820.27  4491.6 1821.07
  4542.1 1818.93  4551.6 1817.28  4571.7 1816.07  4591.7 1816.85  4611.7 1820.03
  4621.7 1820.48  4651.7 1819.12  4731.8 1820.24  4801.8 1819.11  4972.7 1818.43
  4990.4 1810.93  4990.9 1810.43  5011.8 1810.93  5015.2 1814.19  5043.1 1820.51
  5050.4 1821.23  5071.4 1820.99  5128.1 1823.57  5271.7 1822.92    5500 1825.15
#Mann= 3 ,-1 , 0
  3013.4     .05       0  4990.4     .05       0  5011.8     .05       0
Bank Sta=4990.4,5011.8
XS Rating Curve= 0 ,0
Exp/Cntr=0.3,0.1

Type RM Length L Ch R = 1 ,7613    ,179,179,179
BEGIN DESCRIPTION:
Mapping XS 007dd90f
END DESCRIPTION:
XS GIS Cut Line= 5
       1608874.6      6805279.44      1609308.49      6805317.73
      1610205.63      6805428.09      1610418.31      6805577.83
      1610831.41      6805692.46
#Sta/Elev= 30
  3543.4 1821.27  4197.1 1819.77  4270.3 1819.82  4351.5 1820.95  4469.2 1820.24
  4595.3 1821.04  4731.1 1818.41  4741.2 1816.45  4751.3 1815.47  4771.4 1814.87
  4781.5 1815.22  4801.6 1819.64  4831.9 1818.35  4946.4 1819.28    4976  1816.2
  4986.3 1814.02  4986.8 1813.52  5007.2 1813.52  5007.7 1814.02  5011.8 1815.19
  5077.1 1815.41    5098 1817.38  5104.1 1818.94  5126.7 1820.46  5138.8 1822.28
  5181.1 1824.39  5277.1 1824.63  5350.8 1823.25  5532.5 1822.81  5571.7 1823.98
#Mann= 3 ,-1 , 0
  3543.4     .05       0  4986.3     .05       0  5007.7     .05       0
Bank Sta=4986.3,5007.7
XS Rating Curve= 0 ,0
Exp/Cntr=0.3,0.1

Type RM Length L Ch R = 1 ,7434    ,516,516,516
BEGIN DESCRIPTION:
Mapping XS e9dd738d
END DESCRIPTION:
XS GIS Cut Line= 4
      1609169.42      6805434.39      1610088.66      6805577.61
      1610377.72      6805726.05      1610790.87      6805733.84
#Sta/Elev= 30
  3944.2 1820.38  4071.3 1820.46  4133.6 1819.61  4334.4 1818.64  4395.2 1819.16
  4759.5 1819.02  4777.2 1818.61  4789.9 1819.07  4820.2 1819.03    4840 1818.47
  4886.8 1818.31    4909 1817.19  4937.9 1816.94  4947.7  1817.5  4969.9 1815.54
  4972.1 1814.05  4972.6 1813.55    4993 1813.55  4993.5 1814.05  5005.3 1814.83
  5027.8 1814.51  5050.3 1816.28  5095.2 1818.47    5153 1819.06  5169.6  1819.8
  5185.2 1818.94  5199.5 1819.07  5226.8 1820.25  5376.8 1823.16  5612.7 1823.52
#Mann= 3 ,-1 , 0
  3944.2     .05       0  4972.1     .05       0  4993.5     .05       0
Bank Sta=4972.1,4993.5
XS Rating Curve= 0 ,0
Exp/Cntr=0.3,0.1

Type RM Length L Ch R = 1 ,6918    ,640,640,640
BEGIN DESCRIPTION:
Elm 01 91 6918.28
END DESCRIPTION:
XS GIS Cut Line= 3
      1608920.62      6805688.82      1609853.74      6805832.04
      1610825.71      6805792.99
#Sta/Elev= 30
  4058.3  1819.1  4366.2 1819.23  4507.9 1818.05  4745.3 1817.25  4851.9 1817.33
    4877 1817.67  4882.2 1818.25  4922.7 1817.67  4932.8 1816.66  4940.3 1814.47
  4945.4 1814.23    4953 1812.58  4983.4 1811.91  5000.5 1812.15  5002.9 1809.92
  5003.4 1809.42  5023.8 1809.42  5024.3 1809.92  5033.6 1812.98  5043.6 1813.79
  5083.7 1815.65  5093.7 1814.95  5123.7 1816.35  5183.8 1815.82  5343.9 1817.58
    5534 1818.15  5734.2 1822.71  5844.3 1823.43  5924.4 1823.14  5975.1 1823.95
#Mann= 3 ,-1 , 0
  4058.3     .05       0  5002.9     .05       0  5024.3     .05       0
Bank Sta=5002.9,5024.3
XS Rating Curve= 0 ,0
Exp/Cntr=0.3,0.1

Type RM Length L Ch R = 1 ,6278    ,381,381,381
BEGIN DESCRIPTION:
Elm 01 91 6277.69
END DESCRIPTION:
XS GIS Cut Line= 3
      1608944.06      6806246.68      1609874.57      6806274.46
      1610614.15      6806298.76
#Sta/Elev= 30
  4074.3 1817.05  4315.3 1815.27  4365.4 1815.67  4395.4 1814.48  4525.4 1814.21
  4675.5 1812.14  4815.6 1814.75  4855.6  1816.5  4895.6 1815.57  4905.6 1814.47
  4953.5 1812.67  4958.5 1811.86  4965.6  1812.1  4974.9 1808.26  4975.4 1807.76
  4995.8 1807.76  4996.3 1808.26  5002.9 1810.09  5025.7 1811.63  5065.7 1816.08
  5085.7 1816.49  5125.7 1815.58  5275.8 1815.11  5335.8 1815.73  5525.9 1815.77
    5616 1818.45    5656 1818.35    5716 1819.86    5736 1821.24  5745.2 1821.09
#Mann= 3 ,-1 , 0
  4074.3     .05       0  4974.9     .05       0  4996.3     .05       0
Bank Sta=4974.9,4996.3
XS Rating Curve= 0 ,0
Exp/Cntr=0.3,0.1

Type RM Length L Ch R = 1 ,5897    ,258,258,258
BEGIN DESCRIPTION:
Elm 01 91 5898.44
END DESCRIPTION:
XS GIS Cut Line= 4
      1608898.67      6806290.23      1609679.91      6806585.36
      1609805.12      6806586.96      1610581.46      6806628.55
#Sta/Elev= 30
    4049 1817.13  4376.5 1814.61  4399.8 1814.68  4408.5 1815.24  4424.6 1814.08
  4589.7 1811.87  4697.2 1813.75  4884.1 1814.29  4919.2 1814.88  4939.2 1814.34
  4959.2 1811.51  4968.5 1807.73    4969 1807.23  4989.5 1807.23    4990 1807.73
  5006.8 1810.99  5029.3 1812.22  5049.3 1815.04  5069.3 1814.33  5239.6 1813.33
  5269.6 1813.54  5319.7 1815.09  5379.8  1815.9  5419.8 1817.91  5469.9 1817.96
    5520 1819.76  5600.1 1820.14  5650.1 1821.94  5670.2 1821.35  5786.8 1822.33
#Mann= 3 ,-1 , 0
    4049     .05       0  4968.5     .05       0    4990     .05       0
Bank Sta=4968.5,4990
XS Rating Curve= 0 ,0
Exp/Cntr=0.3,0.1

Type RM Length L Ch R = 1 ,5639    ,1595,1595,1595
BEGIN DESCRIPTION:
Mapping XS 93ff9285
END DESCRIPTION:
XS GIS Cut Line= 5
      1608515.38      6806556.93      1609252.39        6806596.
      1609403.44      6806645.48      1609853.96      6806900.68
      1610441.28      6807030.62
#Sta/Elev= 30
    3757 1817.74  3816.7 1816.39  4237.3 1815.72  4467.6 1813.32  4487.6 1813.86
  4493.9 1813.03  4552.7 1811.59  4642.9 1813.24  4816.9 1813.31  4891.9 1814.59
  4920.1 1813.71  4943.1    1814  4956.8 1812.75  4966.1 1814.06  4978.5 1813.32
  4988.6 1811.19  5000.6 1810.31  5005.2 1805.93  5005.7 1805.43  5026.7 1805.93
  5031.9 1809.41  5037.6 1810.56  5066.6 1813.84  5104.1 1814.12    5150  1812.8
  5387.9  1812.5  5531.3 1815.07  5598.5 1817.12  5705.4 1817.64  5773.3 1819.38
#Mann= 5 ,-1 , 0
    3757     .05       0  5005.2     .05       0  5026.7     .05       0
  5066.6     .12       0  5104.1     .05       0
Bank Sta=5005.2,5026.7
XS Rating Curve= 0 ,0
Exp/Cntr=0.3,0.1

Type RM Length L Ch R = 1 ,4044    ,285,285,285
BEGIN DESCRIPTION:
Mapping XS a13c5d73
END DESCRIPTION:
XS GIS Cut Line= 4
      1608533.65      6807145.48      1608994.58      6807291.31
      1609520.62      6807260.06       1610250.8      6807143.13
#Sta/Elev= 30
  4255.9  1815.1  4299.3 1814.02  4379.1 1813.32  4540.5 1813.47  4839.9 1811.93
    4860 1812.05  4882.2 1812.93    4900  1812.5  4930.1  1810.5  4960.2 1809.48
  4980.2 1806.38  4990.2  1806.4  5000.2 1807.19  5009.4 1802.71  5009.9 1802.21
  5030.6 1802.21  5031.1 1802.71  5040.3 1808.44  5060.3 1811.29  5160.5 1812.24
  5180.5 1812.78  5190.6  1813.6  5216.2 1811.78  5370.6  1812.1  5544.2 1809.61
  5696.1 1809.54  5837.9 1811.53  5881.8 1812.44  5918.9 1814.27  6005.8 1815.41
#Mann= 3 ,-1 , 0
  4255.9     .05       0  5009.4     .05       0  5031.1     .05       0
Bank Sta=5009.4,5031.1
XS Rating Curve= 0 ,0
Exp/Cntr=0.3,0.1

Type RM Length L Ch R = 1 ,3759    ,688,688,688
BEGIN DESCRIPTION:
Mapping XS 9552f367
END DESCRIPTION:
XS GIS Cut Line= 4
      1608541.44      6807442.35      1609148.23      6807551.73
      1609489.37      6807489.23      1610335.77      6807166.29
#Sta/Elev= 30
  4173.3 1813.19  4197.2 1812.19  4430.9 1811.82  4516.3 1811.06  4817.1 1810.03
  4888.3 1810.42  4898.6 1811.41  4939.1 1810.28  4969.6 1810.13  4979.7 1808.44
  4989.9 1805.99  4994.1 1801.51  4994.6 1801.01  5015.3 1801.01  5015.8 1801.51
  5020.4 1805.08  5101.7 1811.21  5111.3 1810.88  5164.1 1811.63  5260.4 1810.09
  5381.1 1810.62  5490.7 1809.25  5550.8 1809.39  5624.4 1808.56  5715.3 1809.45
  5752.8 1811.39    5817 1811.86  5885.1 1814.43  5939.9 1814.73  6042.6 1816.71
#Mann= 3 ,-1 , 0
  4173.3     .05       0  4994.1     .05       0  5015.8     .05       0
Bank Sta=4994.1,5015.8
XS Rating Curve= 0 ,0
Exp/Cntr=0.3,0.1

Type RM Length L Ch R = 1 ,3071    ,1785,1785,1785
BEGIN DESCRIPTION:
Mapping XS 3b7e8a69
END DESCRIPTION:
XS GIS Cut Line= 4
      1609257.59      6808124.66      1609387.81      6807799.12
      1609533.64      6807491.83      1610309.69       6807226.2
#Sta/Elev= 30
  4934.8 1808.77  4944.3 1809.74  4968.6 1807.01  4985.1 1803.98  4987.3 1798.76
  4987.8 1798.26  5008.5 1798.26    5009 1798.76    5017 1803.94  5022.4 1805.71
  5038.9 1805.46  5070.9 1807.94  5076.3 1807.56    5082 1808.19  5124.7 1808.55
  5130.1  1809.1  5178.6 1809.33  5356.1 1809.19  5515.1 1810.33  5597.9 1810.42
  5658.7 1811.38  5710.4 1809.96  5859.5 1810.31  6070.9 1808.29  6155.5 1809.31
  6218.9 1811.78  6268.4 1811.65  6299.7 1812.33  6345.7 1814.36  6445.8 1815.38
#Mann= 5 ,-1 , 0
  4934.8     .05       0  4987.3     .05       0    5009     .05       0
  5356.1     .12       0  5515.1     .05       0
Bank Sta=4987.3,5009
XS Rating Curve= 0 ,0
Exp/Cntr=0.3,0.1

Type RM Length L Ch R = 1 ,1286    ,433,433,433
BEGIN DESCRIPTION:
Mapping XS 5420630f
END DESCRIPTION:
XS GIS Cut Line= 4
      1609369.56      6808252.25      1609963.33      6808260.06
      1610429.48      6807898.08      1610676.09      6807451.57
#Sta/Elev= 30
  4039.5 1807.04    4365 1805.56  4657.8 1805.01  4757.3  1805.1  4813.5 1805.91
  4892.2 1805.69  4906.7 1806.31  4927.5 1805.62    4942 1803.71  4977.3 1801.36
  4999.9 1798.13  5003.5 1796.22    5004 1795.72  5024.8 1795.72  5025.3 1796.22
  5035.2 1802.64  5041.5 1803.21    5056 1805.75  5064.2 1806.51  5099.5 1806.94
  5134.8  1806.5  5427.5 1807.16  5486.4 1808.04  5520.6 1809.34  5566.3  1809.5
  5601.6 1811.88  5633.7 1811.71  5661.2 1812.73    5692 1814.82  5733.6 1815.17
#Mann= 3 ,-1 , 0
  4039.5     .05       0  5003.5     .05       0  5025.3     .05       0
Bank Sta=5003.5,5025.3
XS Rating Curve= 0 ,0
Exp/Cntr=0.3,0.1

Type RM Length L Ch R = 1 ,853     ,429,429,429
BEGIN DESCRIPTION:
Mapping XS d848157d
END DESCRIPTION:
XS GIS Cut Line= 4
      1609369.58       6808348.6      1609971.14      6808338.18
      1610351.35      6808444.95      1610468.57      6808421.51
#Sta/Elev= 30
  4103.9  1806.5  4499.4 1805.95  4699.4 1805.04  4792.4 1805.53    4803 1804.47
  4831.7 1804.23  4844.6 1803.47  4865.4 1799.77  4870.9 1800.18  4876.1  1799.6
  4944.3 1799.97  4958.8 1799.43  4978.3 1797.04  4983.5 1797.83  4989.5 1794.72
    4990 1794.22  5010.8 1794.22  5011.3 1794.72  5012.2 1795.46  5017.6 1799.92
  5019.8 1800.73  5031.5 1804.31  5041.9 1805.17  5062.7 1804.45    5091 1804.63
  5104.9 1804.23  5160.8 1804.98  5165.9  1805.8  5175.6 1806.08    5220 1805.84
#Mann= 5 ,-1 , 0
  4103.9     .05       0  4989.5     .05       0  5011.3     .05       0
  5012.2     .12       0  5019.8     .05       0
Bank Sta=4989.5,5011.3
XS Rating Curve= 0 ,0
Exp/Cntr=0.3,0.1

Type RM Length L Ch R = 1 ,424     ,402,402,402
BEGIN DESCRIPTION:
Mapping XS 54f5c4eb
END DESCRIPTION:
XS GIS Cut Line= 4
      1609364.38      6808520.48      1609874.79      6808757.45
      1610288.85      6808653.29      1610624.75      6808619.44
#Sta/Elev= 30
  4252.2 1805.32  4424.1 1805.14  4627.7 1803.83  4887.3 1803.17  4928.6 1803.42
  4938.9 1803.98  4949.2  1801.9  4960.4 1797.62  4969.8 1797.17  4980.1 1795.77
  4985.4  1791.5  4985.9    1791  5006.8    1791  5007.3  1791.5  5011.1 1797.32
  5031.7 1798.96  5052.3 1798.53  5062.6  1798.9  5072.9 1800.26  5078.6 1801.93
  5093.6 1802.86  5114.2  1802.4  5119.7 1804.04  5124.9 1804.48  5160.8 1802.88
  5318.4 1803.73  5338.5 1803.05  5408.9 1805.05  5489.3  1804.9  5579.5 1805.98
#Mann= 3 ,-1 , 0
  4252.2     .05       0  4985.4     .05       0  5007.3     .05       0
Bank Sta=4985.4,5007.3
XS Rating Curve= 0 ,0
Exp/Cntr=0.3,0.1

Type RM Length L Ch R = 1 ,22      ,0,0,0
BEGIN DESCRIPTION:
Elm 01 91 10406.645
END DESCRIPTION:
XS GIS Cut Line= 5
      1609333.11      6808559.53      1610109.19      6809046.69
      1610304.58      6809015.99      1610475.45      6808885.48
      1610760.08      6808705.45
#Sta/Elev= 30
  3885.9 1805.19  4306.8  1803.2  4741.5 1802.24  4802.2 1802.28  4824.6 1803.52
  4868.8 1803.31  4899.2 1802.08  4939.7 1797.74  4954.9 1794.94  4959.9 1796.35
  4970.1  1796.7  4977.6 1790.43  4978.6 1789.93  5017.7 1790.43  5020.4 1796.94
  5055.8 1799.03  5063.4 1800.04  5070.3 1802.24  5076.6 1802.35  5091.1 1804.29
  5113.8 1805.48  5120.2 1805.48  5126.5 1804.09  5133.2 1804.55  5184.6 1803.33
  5241.2 1803.12  5344.6  1804.7  5502.3 1804.54  5532.9 1805.47  5551.8 1805.25
#Mann= 4 ,-1 , 0
  3885.9     .05       0  4977.6     .07       0  5017.7     .05       0
  5133.2     .05       0
Bank Sta=4977.6,5017.7
XS Rating Curve= 0 ,0
Exp/Cntr=0.3,0.1

Chan Stop Cuts=-1
Use User Specified Reach Order=0
Composite Channel Slope=5
