--- Elm 02 01.prj (project) ---

Proj Title=Elm 02 01 Base Level Engineering
Current Plan=p01
Default Exp/Contr=0.3,0.1
English Units
Geom File=g01
Flow File=f01
Plan File=p01
Y Axis Title=Elevation
X Axis Title(PF)=Main Channel Distance
X Axis Title(XS)=Station
BEGIN DESCRIPTION:
Elm 02 01
END DESCRIPTION:
DSS Export Rating Curves= 0
DSS Export Rating Curve Sorted= 0
DSS Export Volume Flow Curves= 0
DXF OffsetX= 0
DXF OffsetY= 0
DXF ScaleX= 1
DXF ScaleY= 10

--- Elm 02 01.p01 (plan) ---

Plan Title=Multiple Run
Short Identifier=Multiple
Geom File=g01
Flow File=f01
Subcritical Flow
K Sum by GR= 0
Std Step Tol= 0.01
Critical Tol= 0.01
Num of Std Step Trials= 20
Max Error Tol= 0.3
Flow Tol Ratio= 0.001
Split Flow NTrial= 30
Split Flow Tol= 0.02
Split Flow Ratio= 0.02
Log Output Level= 0
Friction Slope Method= 1
Unsteady Friction Slope Method= 2
Unsteady Bridges Friction Slope Method= 1
Parabolic Critical Depth
Global Vel Dist=  1 , 1 , 1
Global Log Level= 0
CheckData=True
Encroach Param= -1, 0, 0, 0
BEGIN DESCRIPTION:
Multiple Run
END DESCRIPTION:

--- Elm 02 01.f01 (steady flow) ---

Flow Title=Multiple
Number of Profiles=7
Profile Names=10-year,25-year,50-year,1pct_min,100-year,1pct_plu,500-year
River Rch & RM= Elm 02 01,Reach-1,25016
     201     275     334     252     404     556     600
River Rch & RM= Elm 02 01,Reach-1,18832
     205     280     340     256     410     564     605
River Rch & RM= Elm 02 01,Reach-1,15433
     348     490     608     467     748    1030    1150
River Rch & RM= Elm 02 01,Reach-1,14452
     514     736     925     719    1150    1580    1810
River Rch & RM= Elm 02 01,Reach-1,3549
     576     828    1040     813    1300    1790    2060
Boundary for River Rch & Prof#=Elm 02 01,Reach-1,1
Up Type=0
Dn Type=3
Dn Slope=0.001
Boundary for River Rch & Prof#=Elm 02 01,Reach-1,2
Up Type=0
Dn Type=3
Dn Slope=0.001
Boundary for River Rch & Prof#=Elm 02 01,Reach-1,3
Up Type=0
Dn Type=3
Dn Slope=0.001
Boundary for River Rch & Prof#=Elm 02 01,Reach-1,4
Up Type=0
Dn Type=3
Dn Slope=0.001
Boundary for River Rch & Prof#=Elm 02 01,Reach-1,5
Up Type=0
Dn Type=3
Dn Slope=0.001
Boundary for River Rch & Prof#=Elm 02 01,Reach-1,6
Up Type=0
Dn Type=3
Dn Slope=0.001
Boundary for River Rch & Prof#=Elm 02 01,Reach-1,7
Up Type=0
Dn Type=3
Dn Slope=0.001

--- Elm 02 01.g01 (geometry) ---

Geom Title=Existing Conditions
Program Version=4.10

River Reach=Elm 02 01       ,Reach-1
Reach XY= 30
        1615555.        6823288.      1613906.25      6822934.64
      1613744.53      6822488.93      1610956.01      6822334.39
      1611154.82      6822122.92      1611007.31      6821843.08
      1610665.15      6821937.07      1609665.11      6821597.43
      1609601.38       6820639.5       1608314.8      6819538.71
      1607711.48      6820230.31      1607213.48      6820240.63
      1607044.66      6820698.24      1606812.36      6820731.57
      1607291.88      6820974.78      1607301.47      6821336.53
      1606803.53      6821784.54      1606409.99        6821693.
      1606307.45      6822382.53       1605638.2      6822454.42
      1605614.71      6823077.25       1604610.4      6823035.29
      1604702.62      6823932.47      1604158.33       6824589.7
      1604253.79      6824928.41      1603999.38      6825332.38
      1603305.02      6825680.92      1602610.85      6825340.06
      1602060.41      6825643.17        1601955.        6825988.

Type RM Length L Ch R = 1 ,25016   ,237,237,237
BEGIN DESCRIPTION:
Elm 02 01 24901.344
END DESCRIPTION:
XS GIS Cut Line= 3
      1615507.96      6822863.91      1615506.67      6823288.31
      1615537.04      6823606.97
#Sta/Elev= 30
  4575.6  1835.8  4659.7 1835.26  4699.7 1835.63  4729.7 1835.33  4769.7 1835.48
  4809.7 1834.92  4819.7 1835.12  4839.7 1834.68  4879.7 1834.47  4909.7 1834.47
  4919.7 1834.72  4959.7 1834.55  4995.3 1833.47  4995.6 1832.97  4999.1 1832.97
  4999.3 1833.47  5019.8 1833.85  5029.8 1834.66  5034.9 1835.75    5040 1835.24
  5049.9 1836.42    5060 1836.48    5080 1837.08  5090.1 1837.17  5110.2 1837.99
  5120.2 1838.69  5137.9 1838.37  5180.5 1839.19  5245.8 1839.14  5320.1 1839.87
#Mann= 3 ,-1 , 0
  4575.6     .05       0  4995.3     .03       0  4999.3     .05       0
Bank Sta=4995.3,4999.3
XS Rating Curve= 0 ,0
Exp/Cntr=0.3,0.1

Type RM Length L Ch R = 1 ,24779   ,250,250,250
BEGIN DESCRIPTION:
Elm 02 01 24778.92
END DESCRIPTION:
XS GIS Cut Line= 3
      1615295.87      6822804.79      1615300.21      6823197.55
      1615443.44      6823629.44
#Sta/Elev= 30
  4613.2 1834.19  4726.4 1833.61  4776.4 1833.07  4856.4 1833.08  4936.4 1832.59
  4966.4 1832.79  4984.4 1832.51  4989.4 1832.89    5015  1832.3  5015.2  1831.8
  5018.7  1831.8    5019  1832.3  5027.5 1832.45  5034.9 1832.98  5048.6 1832.83
  5098.3 1834.26  5103.6 1833.97    5130 1834.65  5135.3 1834.59  5143.4 1835.13
  5161.7  1835.3    5167 1835.78  5193.4 1836.25  5206.6 1836.84    5262 1837.83
  5269.8 1838.54  5288.4 1838.87  5293.7 1839.17  5388.8 1839.06    5461  1839.4
#Mann= 3 ,-1 , 0
  4613.2     .05       0    5015     .05       0    5019     .05       0
Bank Sta=5015,5019
XS Rating Curve= 0 ,0
Exp/Cntr=0.3,0.1

Type RM Length L Ch R = 1 ,24529   ,277,277,277
BEGIN DESCRIPTION:
Elm 02 01 24528.54
END DESCRIPTION:
XS GIS Cut Line= 3
      1615141.79      6822728.78       1615089.7      6823078.19
      1615057.15        6823599.
#Sta/Elev= 30
  4653.7 1833.84  4673.1 1833.31  4731.2 1832.51  4736.3  1832.3  4800.5 1832.17
  4805.6 1831.93    4845 1832.08  4855.1 1831.96  4869.8  1832.2  4925.9 1832.08
  4946.1 1831.75  4956.2 1831.88  4976.5 1831.77  4986.6 1831.92  4994.7 1831.15
  4994.9 1830.65  4998.4 1830.65  4998.7 1831.15    5006 1832.14  5009.4 1832.14
  5016.8 1832.53  5026.8 1831.72  5076.9 1831.78    5117 1832.43  5162.3 1832.91
  5167.3 1832.74  5217.2  1833.4  5357.5 1834.12  5397.5 1834.19  5528.8 1834.99
#Mann= 3 ,-1 , 0
  4653.7     .05       0  4994.7     .05       0  4998.7     .05       0
Bank Sta=4994.7,4998.7
XS Rating Curve= 0 ,0
Exp/Cntr=0.3,0.1

Type RM Length L Ch R = 1 ,24252   ,401,401,401
BEGIN DESCRIPTION:
Elm 02 01 24252.45
END DESCRIPTION:
XS GIS Cut Line= 3
      1614885.05       6822733.3       1614847.3      6823041.84
      1614774.39      6823458.47
#Sta/Elev= 30
  4692.5 1831.92  4707.3 1832.16  4717.4 1831.42  4727.5 1831.18  4738.3 1830.38
  4767.8 1830.48    4798 1830.28  4808.1 1830.42  4814.8 1830.21  4819.8 1830.62
  4848.4 1830.42  4858.4 1830.16  4878.6 1830.58  4901.3 1830.46  4949.1 1830.73
  4959.2 1830.48  4969.3 1830.73  4977.7 1830.57  4987.4 1830.05  4987.6 1829.55
  4991.1 1829.55  4991.4 1830.05  5060.4 1830.39  5099.8 1830.89  5182.2 1830.91
  5263.4 1831.27  5278.2 1831.12  5332.6 1831.62  5337.6  1831.5  5426.3  1831.9
#Mann= 3 ,-1 , 0
  4692.5     .05       0  4987.4     .05       0  4991.4     .05       0
Bank Sta=4987.4,4991.4
XS Rating Curve= 0 ,0
Exp/Cntr=0.3,0.1

Type RM Length L Ch R = 1 ,23851   ,369,369,369
BEGIN DESCRIPTION:
Elm 02 01 23851.18
END DESCRIPTION:
XS GIS Cut Line= 3
      1614502.24      6822743.72      1614489.23      6822991.06
      1614495.74      6823360.82
#Sta/Elev= 30
  4754.1 1829.76  4768.4 1830.11  4778.4 1830.11  4795.1 1829.27  4818.5 1829.32
  4828.5 1828.92  4838.5 1829.18  4858.5 1828.98  4868.5 1828.69  4898.6 1828.67
  4918.6 1828.22  4938.6 1828.38  4958.7 1828.12  4968.7 1827.85  4978.7 1826.27
  4983.4 1825.96  4983.6 1825.46  4987.1 1825.46  4987.4 1825.96  4997.8 1826.31
  5008.7 1826.28  5018.7 1826.56  5028.7 1827.56  5038.7 1827.73  5044.8 1828.15
  5049.8 1828.09  5058.7 1828.46  5118.7 1828.22  5168.8 1828.62  5371.6 1829.04
#Mann= 3 ,-1 , 0
  4754.1     .05       0  4983.4     .05       0  4987.4     .05       0
Bank Sta=4983.4,4987.4
XS Rating Curve= 0 ,0
Exp/Cntr=0.3,0.1

Type RM Length L Ch R = 1 ,23482   ,132,132,132
BEGIN DESCRIPTION:
Elm 02 01 23481.93
END DESCRIPTION:
XS GIS Cut Line= 4
      1614314.39      6822715.48      1614172.28      6822841.32
      1614186.38      6822911.85      1614455.52       6823307.8
#Sta/Elev= 30
  4741.1 1828.75  4770.6 1828.15  4778.1 1828.47  4792.4 1827.83    4799 1828.16
  4841.7 1827.46  4870.1 1827.56  4947.9 1826.94  4958.1 1827.32  4966.8 1827.08
  4978.5 1825.09  4986.7 1824.74    4987 1824.24  4990.5 1824.24  4990.7 1824.74
  4998.3  1825.8  5002.8  1825.8  5006.8 1825.06  5012.8 1825.99  5021.7 1825.74
  5034.5 1827.77  5042.7 1828.62  5057.6 1827.14  5070.7 1826.73  5093.5  1826.8
  5120.6 1827.69  5135.5 1827.48  5143.3 1827.03  5192.4 1827.08  5481.6 1828.68
#Mann= 3 ,-1 , 0
  4741.1     .05       0  4986.7     .05       0  4990.7     .05       0
Bank Sta=4986.7,4990.7
XS Rating Curve= 0 ,0
Exp/Cntr=0.3,0.1

Type RM Length L Ch R = 1 ,23350   ,69,69,69
BEGIN DESCRIPTION:
Elm 02 01 23350.49
END DESCRIPTION:
XS GIS Cut Line= 5
      1614260.17      6822673.13      1614102.83      6822809.86
      1614072.45      6822910.77      1614076.79       6822973.7
      1614428.87      6823343.62
#Sta/Elev= 30
  4690.3 1828.19  4704.6 1828.49  4725.4 1827.68  4747.3 1827.52  4761.5 1827.85
  4796.7 1827.32  4803.3 1826.78  4860.3 1827.14  4910.5 1826.33  4928.1 1826.79
  4943.5 1826.55  4969.9 1829.25  4976.5    1829  4981.8 1828.04  5000.1 1828.92
  5021.4 1828.74  5051.5 1828.15  5061.5 1827.56  5066.9 1826.62    5076 1827.73
  5083.2 1826.56  5090.1 1827.66  5097.4 1826.52  5104.3 1826.79  5130.6 1826.27
  5130.8 1825.77  5134.3 1825.77  5134.6 1826.27  5387.4 1827.24  5577.9 1828.55
#Mann= 3 ,-1 , 0
  4690.3     .05       0  5130.6     .05       0  5134.6     .05       0
Bank Sta=5130.6,5134.6
XS Rating Curve= 0 ,0
Exp/Cntr=0.3,0.1

Type RM Length L Ch R = 1 ,23281   ,256,256,256
BEGIN DESCRIPTION:
Elm 02 01 23281.36
END DESCRIPTION:
XS GIS Cut Line= 6
      1614240.63      6822638.42      1614073.54      6822782.73
       1614010.6       6822835.9       1614018.2      6822925.96
      1614037.73      6823058.34       1614372.2      6823444.97
#Sta/Elev= 30
  4608.5 1828.08  4612.4 1827.74    4619 1828.14  4626.7 1827.92  4633.3 1828.28
  4647.5 1827.87  4661.8 1828.05  4690.3 1827.27  4696.9 1827.45  4817.6 1826.45
  4846.1 1826.65    4889 1825.57  4903.3 1825.85  4909.4 1825.44  4933.9  1825.8
  4994.1 1825.96  5011.8 1825.36  5016.8 1825.97  5024.3 1826.03  5034.4 1825.57
  5044.6 1826.12  5054.7 1826.18  5072.9 1825.29  5073.1 1824.79  5076.6 1824.79
  5076.9 1825.29  5081.4 1825.86  5095.1 1826.15  5509.2 1827.66  5647.1 1828.63
#Mann= 3 ,-1 , 0
  4608.5     .05       0  5072.9     .05       0  5076.9     .05       0
Bank Sta=5072.9,5076.9
XS Rating Curve= 0 ,0
Exp/Cntr=0.3,0.1

Type RM Length L Ch R = 1 ,23025   ,548,548,548
BEGIN DESCRIPTION:
Elm 02 01 23025.15
END DESCRIPTION:
XS GIS Cut Line= 4
      1614063.21      6822478.41      1613850.54      6822823.46
       1613764.9       6822945.2      1613741.99      6822998.74
#Sta/Elev= 30
  4604.8 1825.59  4610.6 1825.86  4616.4 1825.36  4647.2 1825.34  4653.1 1824.85
  4683.9 1824.85  4689.8 1824.54  4705.2 1825.21  4711.1 1824.62  4720.6 1825.05
  4726.5 1824.22  4741.9 1824.44  4747.7 1824.06  4763.1 1824.46  4784.4 1824.04
  4799.8 1824.14  4857.8  1823.1  4863.6 1822.69  4921.6 1822.17  5009.9 1822.65
  5025.1 1822.56  5029.2 1822.03  5029.5 1821.53    5033 1821.53  5033.2 1822.03
  5060.8  1822.3  5081.7 1823.29  5153.2 1824.59  5198.5 1824.97  5217.2 1825.72
#Mann= 3 ,-1 , 0
  4604.8     .05       0  5029.2     .05       0  5033.2     .05       0
Bank Sta=5029.2,5033.2
XS Rating Curve= 0 ,0
Exp/Cntr=0.3,0.1

Type RM Length L Ch R = 1 ,22477   ,505,505,505
BEGIN DESCRIPTION:
Elm 02 01 22476.69
END DESCRIPTION:
XS GIS Cut Line= 3
      1613551.06      6822087.79      1613585.78      6822541.34
      1613583.99      6822997.06
#Sta/Elev= 30
  4549.7 1829.15    4590 1828.32  4610.1 1828.36  4630.1 1829.04  4640.2 1828.11
  4666.1 1826.67  4710.4 1826.55  4730.4 1827.19  4750.5 1825.51  4770.6 1824.88
  4796.7 1824.76  4820.7  1825.3  4840.8 1823.63  4860.8 1823.39  4870.8 1823.97
  4890.9 1822.57  4927.4 1821.69  4932.5 1821.85  4961.1 1820.91  4989.2 1819.54
  4989.4 1819.04  4992.9 1819.04  4993.2 1819.54  5061.2 1820.95  5161.2 1820.92
  5191.2 1821.21  5281.2 1823.45  5401.2 1823.53  5431.2 1823.84  5460.3 1824.63
#Mann= 3 ,-1 , 0
  4549.7     .05       0  4989.2     .05       0  4993.2     .05       0
Bank Sta=4989.2,4993.2
XS Rating Curve= 0 ,0
Exp/Cntr=0.3,0.1

Type RM Length L Ch R = 1 ,21972   ,566,566,566
BEGIN DESCRIPTION:
Elm 02 01 21972.13
END DESCRIPTION:
XS GIS Cut Line= 3
       1613199.5      6822057.36      1613132.22      6822493.59
      1613052.02      6822983.48
#Sta/Elev= 30
  4564.4 1826.62  4585.3 1826.74  4605.5 1827.27  4628.8 1825.75    4646 1825.29
  4666.2 1824.94    4697  1824.9  4716.8 1825.53  4737.1 1824.29  4777.5  1823.1
    4818 1822.78  4828.4 1823.45  4858.5 1821.97  4878.7 1821.35  4898.9 1821.02
  4929.3 1821.47  4954.7 1818.88  4959.7 1818.98  4969.8 1818.47  5040.7 1818.99
  5204.5 1818.33  5204.8 1817.83  5208.3 1817.83  5208.5 1818.33  5283.8 1819.28
  5334.5  1819.5  5435.8 1820.75    5457  1820.8  5496.6 1821.42  5502.2 1821.97
#Mann= 3 ,-1 , 0
  4564.4     .05       0  5204.5     .05       0  5208.5     .05       0
Bank Sta=5204.5,5208.5
XS Rating Curve= 0 ,0
Exp/Cntr=0.3,0.1

Type RM Length L Ch R = 1 ,21406   ,545,545,545
BEGIN DESCRIPTION:
Elm 02 01 21406.34
END DESCRIPTION:
XS GIS Cut Line= 3
      1612873.98       6822005.3      1612628.75      6822493.59
      1612253.45      6823283.23
#Sta/Elev= 30
    4459 1821.98  4467.7 1822.09  4495.7 1821.28  4540.4 1820.83  4573.8 1820.96
  4596.1 1821.55  4607.5 1820.81  4652.3 1819.33  4707.8 1818.96  4730.1 1819.39
    4758 1817.73  4786.5 1817.25  4876.1 1816.92  4953.4 1817.15  5024.3  1816.9
  5024.6  1816.4  5028.1  1816.4  5028.3  1816.9  5094.5 1817.07  5145.5 1817.68
  5176.4 1817.55  5208.1 1818.06  5253.5 1818.31  5491.8 1818.39  5552.8 1819.02
    5560 1819.47  5588.2 1819.75  5605.4 1819.15  5663.5 1819.06  5879.7 1820.33
#Mann= 3 ,-1 , 0
    4459     .05       0  5024.3    .035       0  5028.3     .05       0
Bank Sta=5024.3,5028.3
XS Rating Curve= 0 ,0
Exp/Cntr=0.3,0.1

Type RM Length L Ch R = 1 ,20861   ,411,411,411
BEGIN DESCRIPTION:
Elm 02 01 20860.53
END DESCRIPTION:
XS GIS Cut Line= 3
      1612478.84      6821724.62      1612099.05      6822436.45
      1611767.03      6823202.49
#Sta/Elev= 30
  4199.5 1820.54  4263.2 1819.35  4301.5 1819.14  4339.3 1819.62    4351 1818.76
  4455.2 1816.86  4581.2  1816.1  4701.6    1816  4713.4 1815.74  4994.7 1815.41
    4995 1814.91  4998.5 1814.91  4998.7 1815.41  5201.9 1815.93  5215.1 1816.23
  5225.4  1816.2  5230.8 1815.84  5254.3  1816.3  5259.7 1815.69  5487.5 1816.45
  5520.2    1816  5528.8  1816.1  5534.3 1816.65  5610.2 1817.17  5640.1 1818.34
  5672.8  1817.9  5727.3 1818.12  5808.8    1819  5832.3 1819.59  5841.2 1819.37
#Mann= 3 ,-1 , 0
  4199.5     .05       0  4994.7     .05       0  4998.7     .05       0
Bank Sta=4994.7,4998.7
XS Rating Curve= 0 ,0
Exp/Cntr=0.3,0.1

Type RM Length L Ch R = 1 ,20450   ,492,492,492
BEGIN DESCRIPTION:
Elm 02 01 20450.09
END DESCRIPTION:
XS GIS Cut Line= 3
      1612101.21      6821676.93      1611795.23      6822436.45
      1611497.93      6823048.42
#Sta/Elev= 30
  4187.6  1819.7    4222  1820.1  4265.5 1818.68  4414.2 1816.47  4485.2 1815.63
  4512.8 1812.93    4513 1812.43  4516.5 1812.43  4516.8 1812.93    4523 1813.75
  4550.1 1814.49  4592.6 1814.66  4598.4 1814.03    4623 1813.89  4738.6 1814.37
  4753.8 1813.81  4831.7 1814.37  4861.2 1813.91    4868 1814.43  4939.1 1814.57
  4963.3  1814.1  4975.8 1814.63  4992.8 1814.13  5106.3  1814.4  5230.5 1813.53
  5308.3    1815  5352.8 1814.63  5410.7 1815.11  5613.7 1817.12  5686.8 1818.38
#Mann= 7 ,-1 , 0
  4187.6     .05       0  4265.5     .12       0  4414.2     .05       0
  4512.8     .03       0  4516.8     .05       0  4550.1     .12       0
    4623     .05       0
Bank Sta=4512.8,4516.8
XS Rating Curve= 0 ,0
Exp/Cntr=0.3,0.1

Type RM Length L Ch R = 1 ,19958   ,117,117,117
BEGIN DESCRIPTION:
Elm 02 01 19957.98
END DESCRIPTION:
XS GIS Cut Line= 3
      1611375.61      6821583.21      1611379.95      6822394.89
      1611408.12      6822953.89
#Sta/Elev= 30
  4194.2 1814.35    4289 1813.36    4429 1812.86    4469 1812.33    4499 1812.52
    4519 1811.93    4549 1812.18    4579 1811.79    4639 1812.04    4877 1811.39
  4877.2 1810.89  4880.7 1810.89    4881 1811.39    4959 1812.21    4969 1811.44
    4989 1812.62  5010.4 1812.96    5029 1812.25    5039 1812.24  5049.1 1812.73
  5079.1 1812.57  5099.1 1812.98  5159.2  1812.3  5319.4 1814.86  5379.5 1815.18
  5389.5 1814.94  5399.4 1815.31  5404.4 1814.94  5459.6 1816.26  5565.6 1817.18
#Mann= 3 ,-1 , 0
  4194.2     .05       0    4877     .03       0    4881     .05       0
Bank Sta=4877,4881
XS Rating Curve= 0 ,0
Exp/Cntr=0.3,0.1

Type RM Length L Ch R = 1 ,19841   ,388,388,388
BEGIN DESCRIPTION:
Elm 02 01 19840.54
END DESCRIPTION:
XS GIS Cut Line= 3
      1611212.85      6821618.01      1611262.76      6822392.72
      1611260.59       6822920.1
#Sta/Elev= 30
  4228.1 1812.04  4348.3 1810.86  4418.5  1811.2  4528.7 1810.63  4538.7 1811.02
  4608.9  1810.7  4647.1 1810.75    4659 1811.13  4709.1 1810.74  4719.1 1811.12
  4869.4    1811  4899.5 1810.14  4909.5  1810.7  4939.6  1809.9  4969.6 1810.31
  4977.6  1809.7  4977.9  1809.2  4981.4  1809.2  4981.6  1809.7  4999.5 1810.54
  5049.7 1810.08  5069.7  1810.3  5089.7 1810.68  5109.7 1811.64  5199.7 1813.78
  5229.7  1813.8  5409.7 1816.13  5439.7 1816.02  5509.7 1817.03  5531.8 1816.91
#Mann= 3 ,-1 , 0
  4228.1     .05       0  4977.6     .03       0  4981.6     .05       0
Bank Sta=4977.6,4981.6
XS Rating Curve= 0 ,0
Exp/Cntr=0.3,0.1

Type RM Length L Ch R = 1 ,19453   ,621,621,621
BEGIN DESCRIPTION:
Elm 02 01 19453.49
END DESCRIPTION:
XS GIS Cut Line= 6
      1611188.66      6821610.45       1611212.1      6822224.99
      1611139.07      6822227.79      1611002.35      6822284.21
      1610909.03      6822288.55      1610301.42      6822444.79
#Sta/Elev= 30
  4073.9 1811.64  4231.6 1810.66  4291.6 1811.12  4311.6 1810.54  4681.9 1810.65
    4706    1810    4736 1810.09    4746 1812.51  4761.5 1813.98  4833.6  1813.7
  4839.3 1813.27  4910.5 1814.47  4937.9 1813.58  4987.9 1808.94    4996 1807.61
  4996.2 1807.11  4999.7 1807.11    5000 1807.61  5028.7 1810.25  5111.3 1811.03
  5121.7 1810.59  5152.6 1811.27  5180.4 1810.92  5235.2 1811.61  5261.9 1810.56
  5317.8 1811.83  5359.1 1811.02  5384.1 1811.86  5617.3 1812.55  5631.3 1813.22
#Mann= 3 ,-1 , 0
  4073.9     .05       0    4996     .03       0    5000     .05       0
Bank Sta=4996,5000
XS Rating Curve= 0 ,0
Exp/Cntr=0.3,0.1

Type RM Length L Ch R = 1 ,18832   ,421,421,421
BEGIN DESCRIPTION:
Elm 02 01 18831.62
END DESCRIPTION:
XS GIS Cut Line= 3
      1611144.06      6821624.81      1611026.87       6821865.7
      1610534.67      6822286.29
#Sta/Elev= 30
  4735.2 1811.21  4872.2 1809.83  4907.8 1809.76  4924.8 1810.28  4930.4 1809.87
  4947.3 1809.76  4961.2 1808.77  4969.9 1807.83  4975.5 1806.75  4983.4 1806.43
  4992.4 1806.37  5001.6 1807.28  5105.4 1807.34  5154.8 1808.06  5197.7 1807.87
  5310.7 1808.73  5339.3 1808.32  5388.7 1808.56  5408.6 1806.37  5408.8 1805.87
  5412.4 1805.87  5412.7 1806.37  5417.2 1808.13  5431.5 1808.38  5502.9 1809.03
  5517.1 1809.48  5552.2 1809.25  5558.8 1809.69  5580.8 1809.53  5650.5 1810.29
#Mann= 3 ,-1 , 0
  4735.2     .05       0  5408.6     .05       0  5412.7     .05       0
Bank Sta=5408.6,5412.7
XS Rating Curve= 0 ,0
Exp/Cntr=0.3,0.1

Type RM Length L Ch R = 1 ,18411   ,456,456,456
BEGIN DESCRIPTION:
Elm 02 01 18411.36
END DESCRIPTION:
XS GIS Cut Line= 3
      1610959.18      6821536.25      1610647.96      6821932.11
      1610317.22      6822321.44
#Sta/Elev= 30
  4498.4 1809.49  4758.7 1807.92  4793.9 1807.15  4816.5 1807.45  4830.9  1806.9
    4887 1806.36  5000.3 1805.81  5022.8  1806.3  5050.4 1806.28    5056 1805.42
  5056.3 1804.92  5059.9 1804.92  5060.1 1805.42  5064.7  1806.6  5072.4 1806.39
  5078.9  1807.1  5107.5 1807.61  5142.6 1807.48  5185.5 1808.12  5199.8 1807.87
  5249.2 1808.53  5277.7 1808.43  5377.1 1809.35  5384.3 1809.84  5427.1 1809.43
  5441.4 1810.22    5448 1809.91  5483.1 1810.44  5490.8 1810.95  5512.8 1810.92
#Mann= 3 ,-1 , 0
  4498.4     .05       0    5056     .05       0  5060.1     .05       0
Bank Sta=5056,5060.1
XS Rating Curve= 0 ,0
Exp/Cntr=0.3,0.1

Type RM Length L Ch R = 1 ,17955   ,355,355,355
BEGIN DESCRIPTION:
Elm 02 01 17954.53
END DESCRIPTION:
XS GIS Cut Line= 3
      1610604.11      6821407.12      1610416.41      6821748.88
      1610135.37      6822162.29
#Sta/Elev= 30
  4611.2  1806.9  4831.1 1805.48    4869 1806.11  4897.4 1805.85  4920.2 1804.91
  4988.3 1804.63  4997.8 1804.17  5009.3 1804.24  5013.3 1803.44  5013.5 1802.94
  5017.1 1802.94  5017.4 1803.44  5024.2 1804.02  5036.3 1806.04  5045.2 1806.27
  5087.2  1806.1  5096.1 1806.62    5132 1806.65  5145.2 1806.23  5245.8 1806.72
  5281.8 1807.34  5302.7 1807.07  5311.6 1807.63  5353.6 1807.43  5368.6 1807.93
  5398.4 1807.24  5404.5 1807.46  5411.2 1808.39  5425.5 1808.09    5501  1808.9
#Mann= 3 ,-1 , 0
  4611.2     .05       0  5013.3     .05       0  5017.4     .05       0
Bank Sta=5013.3,5017.4
XS Rating Curve= 0 ,0
Exp/Cntr=0.3,0.1

Type RM Length L Ch R = 1 ,17600   ,416,416,416
BEGIN DESCRIPTION:
Elm 02 01 17599.32
END DESCRIPTION:
XS GIS Cut Line= 5
       1610552.2      6821349.85        1610142.      6821506.11
      1610128.79      6821640.66      1610130.62      6821890.21
      1610072.92       6822114.5
#Sta/Elev= 30
  4428.1 1806.82  4488.5 1806.52  4608.9 1804.88  4778.8 1804.48  4862.8 1803.66
  4979.5 1804.19  4992.2  1803.8  4998.4 1802.55  5002.2 1802.55  5007.5 1801.79
  5007.8 1801.29  5011.4 1801.29  5011.6 1801.79  5029.6 1803.22  5039.6 1803.39
  5069.6 1802.91  5089.6 1803.87  5109.6  1803.7  5119.6 1803.16  5189.6 1805.12
  5254.5 1806.35  5301.2 1806.47  5330.8 1807.27  5335.9  1806.6  5352.8 1807.34
  5376.7 1806.54  5394.1 1807.59  5445.7  1808.3  5452.9 1807.86  5483.4 1808.34
#Mann= 3 ,-1 , 0
  4428.1     .05       0  5007.5     .05       0  5011.6     .05       0
Bank Sta=5007.5,5011.6
XS Rating Curve= 0 ,0
Exp/Cntr=0.3,0.1

Type RM Length L Ch R = 1 ,17184   ,471,471,471
BEGIN DESCRIPTION:
Elm 02 01 17290.47
END DESCRIPTION:
XS GIS Cut Line= 4
      1610573.86      6821291.27      1609972.32      6821426.82
       1609777.2      6821769.26      1609605.34      6822232.77
#Sta/Elev= 30
  4035.7 1806.79  4157.5 1806.41  4268.1 1805.02  4456.5 1804.22  4639.7 1802.69
  4688.2 1802.65  4733.2 1803.38  4754.8 1802.98  4760.5 1803.49  4776.4 1803.03
  4813.8 1803.19  4826.3 1803.78  4878.7 1803.02  4906.9 1803.35  4937.7 1802.51
  4943.5 1802.83  5010.5 1802.25  5022.1 1801.18  5022.4 1800.68    5026 1800.68
  5026.3 1801.18  5033.5 1801.39    5040 1802.31  5043.6 1803.54  5055.8 1804.68
  5069.5 1804.89  5099.9 1806.73    5150  1806.2  5387.7 1808.49  5540.8 1807.96
#Mann= 3 ,-1 , 0
  4035.7     .05       0  5022.1     .05       0  5026.3     .05       0
Bank Sta=5022.1,5026.3
XS Rating Curve= 0 ,0
Exp/Cntr=0.3,0.1

Type RM Length L Ch R = 1 ,16713   ,399,399,399
BEGIN DESCRIPTION:
Elm 02 01 16713.68
END DESCRIPTION:
XS GIS Cut Line= 3
      1610580.35      6821258.72      1609790.22      6821378.64
      1609288.49      6821395.81
#Sta/Elev= 30
    4023 1806.84  4317.4 1805.29  4412.8 1804.14  4635.3 1803.03  4655.9 1803.33
  4706.1 1802.86  4736.4 1801.95  4746.5 1802.18  4783.3 1801.58  4822.2  1801.5
  4837.4 1800.26  4847.4 1800.07  4887.4 1800.21  4917.5 1800.95  4951.1 1800.92
  4977.5 1799.88  4987.5 1799.85  4995.4 1799.18  4995.6 1798.68  4999.3 1798.68
  4999.6 1799.18  5007.5 1800.69  5017.5 1801.87  5047.5 1802.52  5087.6 1802.84
  5097.6 1803.36  5137.6 1803.78  5207.6  1805.5  5267.7 1806.03  5324.2    1806
#Mann= 3 ,-1 , 0
    4023     .05       0  4995.4     .05       0  4999.6     .05       0
Bank Sta=4995.4,4999.6
XS Rating Curve= 0 ,0
Exp/Cntr=0.3,0.1

Type RM Length L Ch R = 1 ,16314   ,307,307,307
BEGIN DESCRIPTION:
Elm 02 01 16313.64
END DESCRIPTION:
XS GIS Cut Line= 3
      1610535.28      6821071.51      1609652.77      6821098.99
      1609221.75      6821181.03
#Sta/Elev= 30
  4118.8 1805.97  4279.2 1804.88  4469.3  1804.7  4649.3 1803.74  4669.3  1804.1
  4719.4 1803.17  4859.4 1801.96  4909.5 1800.87  4939.5 1799.28  4949.5 1799.14
  4969.5 1799.75  5001.7 1799.99  5009.6 1799.64    5019 1797.92  5027.9 1797.86
  5028.2 1797.36  5031.9 1797.36  5032.1 1797.86  5050.4 1799.21  5076.2 1798.71
  5081.3 1799.34  5133.5 1799.95  5162.3 1798.72  5172.5    1799  5180.6 1800.09
  5185.7 1800.08  5192.9 1801.16  5213.2 1801.86  5347.4 1805.06  5440.5 1805.24
#Mann= 3 ,-1 , 0
  4118.8     .05       0  5027.9     .05       0  5032.1     .05       0
Bank Sta=5027.9,5032.1
XS Rating Curve= 0 ,0
Exp/Cntr=0.3,0.1

Type RM Length L Ch R = 1 ,16007   ,299,299,299
BEGIN DESCRIPTION:
Elm 02 01 16006.56
END DESCRIPTION:
XS GIS Cut Line= 4
      1610486.66       6820292.5      1609955.45      6820560.84
      1609650.69      6820792.52      1609255.88      6821093.81
#Sta/Elev= 30
    4022 1812.61  4102.3 1810.01  4182.3 1806.29  4303.9  1803.7  4377.4 1802.53
    4416 1802.64    4422 1802.09  4444.2 1801.69  4472.1 1801.81  4550.1 1800.26
  4600.3 1800.06  4606.4 1799.13  4630.3 1799.92  4651.4 1799.12  4680.5 1800.23
  4736.7 1800.89  4886.4 1800.26  4936.3 1799.42  4950.9 1796.46  4963.3 1795.93
  4963.6 1795.43  4967.3 1795.43  4967.6 1795.93  5071.5 1798.94  5129.6 1798.03
  5264.7  1800.6  5285.6 1801.71  5321.6 1802.05  5399.9 1804.35  5496.6 1804.85
#Mann= 3 ,-1 , 0
    4022     .05       0  4963.3     .05       0  4967.6     .05       0
Bank Sta=4963.3,4967.6
XS Rating Curve= 0 ,0
Exp/Cntr=0.3,0.1

Type RM Length L Ch R = 1 ,15708   ,275,275,275
BEGIN DESCRIPTION:
Elm 02 01 16994.478
END DESCRIPTION:
XS GIS Cut Line= 3
      1609890.25       6819883.7      1609513.07      6820544.08
      1609082.99      6820930.53
#Sta/Elev= 30
  4239.5 1801.04  4384.8 1800.63  4414.5 1799.97  4475.6 1799.49  4670.5 1798.53
  4744.7    1796  4760.6 1797.59  4884.4 1796.78  4912.4 1795.96  4943.4 1797.31
  4968.6 1794.21  4968.9 1793.71  4972.6 1793.71  4972.9 1794.21  5002.1 1794.99
  5022.9 1797.04  5072.3 1797.71  5157.5 1800.61  5227.7  1800.5  5241.9 1801.19
  5270.4  1801.1  5298.8 1801.87  5306.2 1803.01    5313 1802.26  5320.1 1804.45
  5341.4  1804.3  5348.1 1804.82  5355.6 1803.94  5525.2 1804.61  5578.2 1804.09
#Mann= 5 ,-1 , 0
  4239.5     .05       0  4414.5     .12       0  4475.6     .05       0
  4968.6     .05       0  4972.9     .05       0
Bank Sta=4968.6,4972.9
XS Rating Curve= 0 ,0
Exp/Cntr=0.3,0.1

Type RM Length L Ch R = 1 ,15433   ,251,251,251
BEGIN DESCRIPTION:
Elm 02 01 15433.09
END DESCRIPTION:
XS GIS Cut Line= 5
      1609577.33      6820105.07      1609422.82      6820202.29
      1609368.04      6820284.21      1609304.22      6820438.28
      1609196.81      6820611.87
#Sta/Elev= 30
  4556.9 1797.61  4647.6 1797.09  4684.1 1796.56  4705.3 1796.72  4735.2 1796.02
  4739.5 1796.02  4742.4 1796.43  4748.4 1796.13  4778.4 1796.43  4858.7 1796.16
  4864.1  1795.8  4917.9 1795.35  4935.8 1794.81  4950.3  1793.8    4972 1793.25
  4979.7 1792.59  4980.2 1792.09  4985.5 1792.09    4986 1792.59  4994.4 1792.96
  5001.9 1793.96  5007.5 1793.96  5011.6 1795.06  5048.2 1797.29  5069.5 1798.23
  5127.4 1799.46  5133.8 1800.04  5148.6 1799.95    5164 1800.52  5208.9 1800.87
#Mann= 3 ,-1 , 0
  4556.9     .05       0  4979.7     .05       0    4986     .05       0
Bank Sta=4979.7,4986
XS Rating Curve= 0 ,0
Exp/Cntr=0.3,0.1

Type RM Length L Ch R = 1 ,15182   ,299,299,299
BEGIN DESCRIPTION:
Elm 02 01 15181.72
END DESCRIPTION:
XS GIS Cut Line= 4
      1609563.45      6820096.39      1609214.48      6820238.75
      1609105.66      6820290.71      1608830.02      6820445.89
#Sta/Elev= 30
  4504.7 1797.63  4507.7 1797.61  4633.1 1796.39  4657.1 1796.51  4681.1 1795.87
  4734.6 1795.77    4773 1795.25  4788.1 1795.48  4812.1 1795.07  4817.5 1795.49
  4848.6 1794.85  4865.6  1795.1    4889 1794.64  4903.2 1793.17  4925.3 1791.68
  4931.2 1791.61  4931.7 1791.11    4937 1791.11  4937.5 1791.61  4939.9 1792.14
  4969.7 1791.72  5004.5 1791.97  5023.7  1793.9  5051.1 1795.55    5067 1795.52
  5088.7 1796.19    5132 1796.65  5228.9 1796.43  5293.9 1797.36  5318.5 1797.01
#Mann= 4 ,-1 , 0
  4504.7     .12       0  4507.7     .05       0  4931.2     .05       0
  4937.5     .05       0
Bank Sta=4931.2,4937.5
XS Rating Curve= 0 ,0
Exp/Cntr=0.3,0.1

Type RM Length L Ch R = 1 ,14883   ,96,96,96
BEGIN DESCRIPTION:
Elm 02 01 14883.48
END DESCRIPTION:
XS GIS Cut Line= 4
      1609539.16        6820020.      1608933.38      6820121.93
      1608848.49       6820182.2      1608672.71      6820346.05
#Sta/Elev= 30
  4283.8 1797.76  4328.6 1797.67  4450.3 1795.91  4484.2 1795.85  4490.8 1795.06
    4501 1794.92    4572 1794.42  4600.3 1794.44  4605.3 1794.87  4612.5 1794.21
  4621.7 1794.03  4774.8 1793.74  4855.9 1794.23  4898.1 1793.22  4901.1 1792.66
    4922 1791.39  4981.1 1790.29  5005.4 1787.77  5005.9 1787.27  5011.3 1787.27
  5011.8 1787.77  5015.9 1788.52  5022.8 1792.08  5030.1 1793.66  5036.9 1794.54
  5164.4 1794.78  5185.4 1795.29  5206.9 1794.99  5227.9 1795.43  5242.5 1795.19
#Mann= 4 ,-1 , 0
  4283.8     .12       0  4621.7     .05       0  5005.4     .05       0
  5011.8     .05       0
Bank Sta=5005.4,5011.8
XS Rating Curve= 0 ,0
Exp/Cntr=0.3,0.1

Type RM Length L Ch R = 1 ,14787   ,335,335,335
BEGIN DESCRIPTION:
Elm 02 01 15042.487
END DESCRIPTION:
XS GIS Cut Line= 4
      1609494.04      6819980.06      1608898.51      6820051.25
      1608551.07      6820236.59      1608508.23      6820343.79
#Sta/Elev= 30
  4292.2 1797.65  4348.6 1797.16  4452.4 1794.83  4472.5 1795.32  4673.9 1794.29
  4694.1 1793.95  4724.3 1792.87  4733.8 1792.07  4738.8 1792.44  4754.5 1791.62
  4826.2 1793.33  4865.3 1793.78  4907.3 1793.59  4920.6 1792.54    4930 1791.04
  4936.9 1789.01  4942.6 1788.34  4997.1 1788.32  5002.8 1788.72  5006.1 1787.63
  5006.6 1787.13    5012 1787.13  5012.5 1787.63  5024.7 1788.09    5032 1790.96
    5041 1791.89  5046.7 1793.16    5063 1793.89  5285.8 1793.73  5401.2 1795.21
#Mann= 4 ,-1 , 0
  4292.2     .12       0  4348.6     .05       0  5006.1     .05       0
  5012.5     .05       0
Bank Sta=5006.1,5012.5
XS Rating Curve= 0 ,0
Exp/Cntr=0.3,0.1

Type RM Length L Ch R = 1 ,14452   ,334,334,334
BEGIN DESCRIPTION:
Elm 02 01 14452.2
END DESCRIPTION:
XS GIS Cut Line= 3
      1608828.28      6819386.43      1608648.61      6819844.73
      1608442.89      6820266.58
#Sta/Elev= 30
  4509.7 1795.53  4543.6 1796.11  4565.1 1794.73  4589.6 1794.07  4673.6 1793.78
  4683.2 1793.15  4692.7 1793.32  4704.7 1792.28  4752.3 1791.81  4769.2 1792.21
  4812.1 1790.68  4898.1 1791.11  4930.3 1790.18  4939.5 1790.52  4944.9 1789.81
  4951.8 1790.72  4974.7 1790.81    4984  1790.2  4993.8 1788.58  4997.6  1785.5
  4998.1    1785  5005.8    1785  5006.3  1785.5  5027.8 1788.48  5044.5 1788.29
  5072.6 1789.45  5112.1 1792.27  5230.3 1791.91    5388 1793.11  5471.3 1794.38
#Mann= 3 ,-1 , 0
  4509.7     .05       0  4997.6     .05       0  5006.3     .05       0
Bank Sta=4997.6,5006.3
XS Rating Curve= 0 ,0
Exp/Cntr=0.3,0.1

Type RM Length L Ch R = 1 ,14118   ,535,535,535
BEGIN DESCRIPTION:
Elm 02 01 14118.32
END DESCRIPTION:
XS GIS Cut Line= 4
      1608580.89      6819351.27      1608450.69       6819637.7
      1608382.78       6819834.2      1608400.25      6820223.07
#Sta/Elev= 30
  4687.9 1793.67  4718.5 1793.43  4736.1 1792.87  4741.6 1793.27  4759.1  1792.6
  4764.6 1792.88  4810.8 1791.96  4839.3 1792.59  4849.1 1791.54  4862.4 1790.84
  4908.5 1790.33    4926 1789.59  4937.1 1787.99  4954.7  1786.7  4955.8 1785.43
  4956.3 1784.93    4964 1784.93  4964.5 1785.43  4969.9 1785.93  5002.5 1787.17
  5013.4 1788.26    5024 1788.71  5063.5 1789.58  5076.9 1789.51  5087.5 1789.96
  5182.7 1790.61  5274.3 1789.99  5334.4 1790.11  5424.5 1790.93  5599.7 1793.89
#Mann= 3 ,-1 , 0
  4687.9     .05       0  4955.8     .05       0  4964.5     .05       0
Bank Sta=4955.8,4964.5
XS Rating Curve= 0 ,0
Exp/Cntr=0.3,0.1

Type RM Length L Ch R = 1 ,13583   ,473,473,473
BEGIN DESCRIPTION:
Elm 02 01 13583.17
END DESCRIPTION:
XS GIS Cut Line= 4
      1607759.97      6819565.58      1608009.94      6819685.35
      1608255.76      6819882.48      1608332.54      6820139.79
#Sta/Elev= 30
    4722 1790.71  4945.6 1790.61  4960.4 1791.52  4973.8 1791.62  4999.2 1790.56
  5005.3 1788.56  5011.7 1788.06  5026.1 1785.01  5036.1 1783.38  5036.6 1782.88
  5044.4 1782.88  5044.9 1783.38    5047 1784.55  5054.9 1785.06  5061.4 1784.87
  5096.6 1786.33  5139.8 1786.53    5175 1787.88  5210.8 1787.89  5261.4 1788.97
  5267.8 1788.58  5310.6 1789.77    5320 1789.39  5327.2 1789.71  5431.8 1789.81
  5445.3 1789.49  5476.6 1790.77  5497.5 1790.43  5549.6 1792.48  5582.8 1793.02
#Mann= 3 ,-1 , 0
    4722     .05       0  5036.1     .05       0  5044.9     .05       0
Bank Sta=5036.1,5044.9
XS Rating Curve= 0 ,0
Exp/Cntr=0.3,0.1

Type RM Length L Ch R = 1 ,13110   ,532,532,532
BEGIN DESCRIPTION:
Elm 02 01 13109.83
END DESCRIPTION:
XS GIS Cut Line= 4
      1607481.83      6819671.02      1607730.48      6819977.46
      1607817.72      6820027.05      1608043.68      6820184.01
#Sta/Elev= 30
  4505.4  1790.2  4527.3 1790.68    4534 1789.87  4548.3 1790.45  4569.2 1789.74
  4577.1 1790.37  4583.5 1789.52  4633.1  1790.3    4641 1789.55  4661.8 1789.68
  4676.2 1788.48  4740.2 1787.36  4804.1 1787.67  4899.6 1786.69    4927 1787.22
  4939.7 1786.43  4948.6 1782.37  4954.3 1785.03  4962.7 1781.34  4981.3 1780.69
  4981.8 1780.19  4990.2 1780.69  4991.8 1783.34  4996.3  1781.4    5007 1782.29
  5013.1  1781.6    5034 1784.56  5048.9 1785.61  5084.7 1785.44  5275.5 1788.97
#Mann= 3 ,-1 , 0
  4505.4     .05       0  4981.3     .05       0  4990.2     .05       0
Bank Sta=4981.3,4990.2
XS Rating Curve= 0 ,0
Exp/Cntr=0.3,0.1

Type RM Length L Ch R = 1 ,12578   ,301,301,301
BEGIN DESCRIPTION:
Elm 02 01 12577.72
END DESCRIPTION:
XS GIS Cut Line= 3
      1607223.97      6819886.42       1607427.1      6820266.63
      1607767.34      6820323.92
#Sta/Elev= 30
  4570.1 1786.98  4673.9 1785.69    4690  1785.1  4696.6 1785.38  4750.1 1784.07
  4777.8 1784.78  4837.9 1784.31  4876.2 1783.47  4934.7 1783.72  4947.7 1783.55
    4964 1782.46    4980 1782.21  4981.5 1781.78    4982 1781.28  4989.9 1781.28
  4990.4 1781.78  4991.6 1782.27  5029.5 1782.52    5037 1781.92  5042.1 1782.84
  5049.7  1783.1  5097.6 1783.77  5102.6 1784.35  5158.1 1785.22  5171.4 1785.92
  5218.6  1785.7  5223.7 1786.31  5252.6 1785.04  5293.1 1787.35  5346.2 1787.77
#Mann= 3 ,-1 , 0
  4570.1     .05       0  4981.5     .05       0  4990.4     .05       0
Bank Sta=4981.5,4990.4
XS Rating Curve= 0 ,0
Exp/Cntr=0.3,0.1

Type RM Length L Ch R = 1 ,12277   ,204,204,204
BEGIN DESCRIPTION:
Elm 02 01 12276.88
END DESCRIPTION:
XS GIS Cut Line= 4
      1607046.88      6819842.99      1607192.72      6820303.09
      1607322.93      6820360.38      1607681.11      6820372.49
#Sta/Elev= 30
  4520.8 1787.93    4547 1787.23  4683.4 1787.59  4724.9 1785.65  4746.4 1786.06
  4756.8 1785.49  4762.4 1783.69  4767.7 1783.61  4809.3 1775.96  4832.3 1774.15
  4859.3 1773.75  4860.1    1773  4860.6  1772.5    4869    1773  4903.7 1775.65
  4914.2 1777.47  4929.1 1778.42  4966.7 1779.77  4993.7 1779.66  4998.9 1782.77
  5025.2 1784.09  5030.7 1783.44  5038.7 1783.78  5048.5 1784.89    5054 1787.64
  5060.6 1788.14  5077.3 1784.52  5106.2 1783.52  5277.9 1786.09  5504.1 1787.58
#Mann= 3 ,-1 , 0
  4520.8     .05       0  4860.1     .05       0    4869     .05       0
Bank Sta=4860.1,4869
XS Rating Curve= 0 ,0
Exp/Cntr=0.3,0.1

Type RM Length L Ch R = 1 ,12073   ,654,654,654
BEGIN DESCRIPTION:
Elm 02 01 12072.88
END DESCRIPTION:
XS GIS Cut Line= 3
      1606498.33      6820488.42      1607055.57      6820450.23
      1607647.55      6820429.39
#Sta/Elev= 30
  4439.9 1784.86  4486.7 1785.09  4515.4 1786.22  4536.8  1785.6  4668.7 1785.17
  4707.2 1784.34  4777.4 1782.08  4857.6 1782.21  4907.7 1781.83  4927.7 1782.33
  4967.8 1782.33  4987.9 1781.52  4995.7 1780.03  5000.7 1780.03  5007.9 1778.88
  5017.9 1778.34  5023.4  1777.5  5023.9    1777  5031.9    1777  5032.4  1777.5
  5047.9 1779.35  5067.9 1781.03  5107.9 1782.59    5168 1783.11    5178 1782.76
    5188 1783.11  5203.4 1782.69    5218 1782.79  5318.1 1785.47  5590.8 1787.17
#Mann= 3 ,-1 , 0
  4439.9     .05       0  5023.4     .05       0  5032.4     .05       0
Bank Sta=5023.4,5032.4
XS Rating Curve= 0 ,0
Exp/Cntr=0.3,0.1

Type RM Length L Ch R = 1 ,11419   ,744,744,744
BEGIN DESCRIPTION:
Elm 02 01 11419.17
END DESCRIPTION:
XS GIS Cut Line= 3
      1606445.83      6820854.91      1606850.36      6820839.29
      1607650.37      6820650.13
#Sta/Elev= 30
  4595.2 1783.62  4664.4 1783.98  4704.4 1783.04  4901.7 1782.46  4924.6 1781.28
  4954.6 1778.24  4964.6 1778.05  4974.6 1775.07  4980.2 1774.99  4980.7 1774.49
  4988.7 1774.49  4989.2 1774.99  4994.7 1777.86  4999.8 1778.65    5005 1778.65
  5028.9 1780.79    5087  1780.1  5148.7 1780.56  5160.9 1779.84  5169.2 1780.85
  5261.7 1781.14  5377.4 1783.42    5385 1783.11  5551.7 1785.33  5600.8 1785.25
  5631.1 1785.93  5636.3 1785.47  5805.4 1787.46  5810.5 1786.98  5822.1  1787.3
#Mann= 3 ,-1 , 0
  4595.2     .05       0  4980.2     .05       0  4989.2     .05       0
Bank Sta=4980.2,4989.2
XS Rating Curve= 0 ,0
Exp/Cntr=0.3,0.1

Type RM Length L Ch R = 1 ,10675   ,303,303,303
BEGIN DESCRIPTION:
Elm 02 01 10674.72
END DESCRIPTION:
XS GIS Cut Line= 3
      1606815.77      6821138.94      1607256.73      6821116.37
      1607775.84      6821081.65
#Sta/Elev= 30
  4560.4    1781  4629.7 1780.39  4669.8 1780.48  4719.8 1779.51  4729.8 1779.81
  4789.9 1779.03    4850 1779.37    4860 1778.97  4960.1  1778.5  5001.9 1777.79
  5010.2 1776.76  5020.2 1774.64  5025.7 1774.37  5026.2 1773.87  5034.3 1773.87
  5034.8 1774.37  5040.3 1776.93  5048.9 1778.89  5060.3 1780.69  5130.5 1784.65
  5160.6 1785.29  5170.6 1786.02    5204 1786.44  5230.7 1786.27  5240.7 1786.77
  5280.8 1786.82    5381 1788.06  5421.1 1788.11  5481.3 1789.22  5522.2 1789.51
#Mann= 3 ,-1 , 0
  4560.4     .05       0  5025.7     .05       0  5034.8     .05       0
Bank Sta=5025.7,5034.8
XS Rating Curve= 0 ,0
Exp/Cntr=0.3,0.1

Type RM Length L Ch R = 1 ,10372   ,439,439,439
BEGIN DESCRIPTION:
Elm 02 01 10372.19
END DESCRIPTION:
XS GIS Cut Line= 3
      1606823.18      6821235.59      1607258.93      6821386.63
      1607654.42      6821553.15
#Sta/Elev= 30
  4540.3 1780.46  4628.1 1779.76  4648.1 1779.05  4716.2 1778.21  4753.9 1776.82
  4773.2 1777.38  4835.5  1777.1  4849.2 1777.54  4880.9 1776.58  4928.9 1777.63
  4934.2 1777.19  4960.1 1777.39  4976.2 1776.02  4991.2 1776.44  5001.5 1775.74
  5003.5 1774.42    5004 1773.92  5012.1 1773.92  5012.6 1774.42  5015.7 1775.37
  5021.1 1775.33  5039.4 1778.87  5121.5 1784.23  5198.1 1785.89  5203.5 1785.54
  5235.9 1786.15  5268.5 1785.94  5280.2 1786.55  5311.9 1786.33  5430.6  1787.7
#Mann= 3 ,-1 , 0
  4540.3     .05       0  5003.5     .05       0  5012.6     .05       0
Bank Sta=5003.5,5012.6
XS Rating Curve= 0 ,0
Exp/Cntr=0.3,0.1

Type RM Length L Ch R = 1 ,9933    ,718,718,718
BEGIN DESCRIPTION:
Elm 02 01 9933.35
END DESCRIPTION:
XS GIS Cut Line= 3
      1606508.91      6821379.67      1606882.19      6821561.97
      1607350.49      6821711.13
#Sta/Elev= 30
  4585.6 1780.47  4747.7 1779.62  4759.3 1779.16  4770.2 1779.43  4803.8 1778.48
  4826.4 1778.54  4881.7  1776.9  4910.9 1777.22  4916.4 1776.83  4926.2 1776.98
  4948.5 1776.49  4961.5 1776.16  4970.8 1773.47  4978.5 1771.75  4979.4 1771.12
  4979.9 1770.62  4988.1 1770.62  4988.6 1771.12  5006.8 1775.39  5014.5 1775.61
  5033.8 1775.96  5056.4  1775.5  5087.9 1775.48  5108.9 1776.06  5213.9 1777.16
  5381.8 1782.85  5403.9 1782.92  5436.1 1783.83  5444.8 1783.62  5492.5 1784.34
#Mann= 3 ,-1 , 0
  4585.6     .05       0  4979.4     .03       0  4988.6     .05       0
Bank Sta=4979.4,4988.6
XS Rating Curve= 0 ,0
Exp/Cntr=0.3,0.1

Type RM Length L Ch R = 1 ,9215    ,399,399,399
BEGIN DESCRIPTION:
Elm 02 01 9215.33
END DESCRIPTION:
XS GIS Cut Line= 3
      1606058.42      6821464.74        1606410.      6821694.79
      1607011.68      6822080.03
#Sta/Elev= 30
  4580.6 1780.68  4754.9 1780.67  4941.8 1778.38    4957 1776.33  4970.9 1775.94
  4993.1 1776.53  4999.1 1773.87  5006.7 1773.29  5009.5  1768.8    5010  1768.3
  5018.6  1768.3  5019.1  1768.8  5020.2 1769.66  5029.5 1770.84  5042.3 1771.13
  5071.8 1773.51    5093 1774.07  5137.3  1774.2  5150.5 1775.06  5180.9 1774.74
  5232.3 1775.21  5238.4 1775.75  5259.5 1775.41  5267.9 1775.92    5317 1775.97
  5353.4 1776.83  5410.9 1776.74  5571.5 1778.29  5665.4 1779.88  5715.2 1781.27
#Mann= 3 ,-1 , 0
  4580.6     .05       0  5009.5     .05       0  5019.1     .05       0
Bank Sta=5009.5,5019.1
XS Rating Curve= 0 ,0
Exp/Cntr=0.3,0.1

Type RM Length L Ch R = 1 ,8816    ,705,705,705
BEGIN DESCRIPTION:
Elm 02 01 8815.6
END DESCRIPTION:
XS GIS Cut Line= 3
      1605928.26      6821874.92        1606410.      6822063.71
       1606940.8      6822152.54
#Sta/Elev= 30
  4487.9 1779.02  4540.5 1778.14  4733.1 1777.92  4811.8  1776.3  4828.1 1776.72
  4950.1 1775.23    4957  1774.9  4967.7 1772.27  4974.5 1768.47  4975.1 1766.81
  4975.6 1766.31  4984.2 1766.31  4984.7 1766.81    4999 1769.53  5010.4 1769.95
  5020.5 1771.58  5040.8 1772.15  5050.9 1771.15  5058.8 1771.37  5063.9 1773.44
  5071.2 1773.78  5172.6 1772.77  5185.3 1772.07  5192.9 1770.84  5223.3 1771.25
  5253.7 1774.04  5294.3 1776.13  5301.7 1777.58  5385.5 1777.78  5543.5 1781.29
#Mann= 3 ,-1 , 0
  4487.9     .05       0  4975.1     .05       0  4984.7     .05       0
Bank Sta=4975.1,4984.7
XS Rating Curve= 0 ,0
Exp/Cntr=0.3,0.1

Type RM Length L Ch R = 1 ,8111    ,563,563,563
BEGIN DESCRIPTION:
Elm 02 01 8110.98
END DESCRIPTION:
XS GIS Cut Line= 3
      1605660.77      6822026.83      1606023.18       6822391.4
      1606370.22      6822836.05
#Sta/Elev= 30
  4490.7  1778.1  4551.1 1777.84  4558.2 1776.57  4565.2 1777.47  4572.3 1776.21
  4579.4 1777.43  4586.5 1776.06  4593.5 1777.21  4600.6 1775.51  4607.6  1776.7
  4614.7 1775.22  4621.8 1776.38  4628.9 1774.81  4635.9 1775.44    4643 1774.53
  4671.3 1774.66  4734.9 1773.21  4770.3 1771.57    4841 1770.97  4890.5 1768.94
  4968.3 1769.46  5004.8 1765.78  5006.4  1763.3  5006.9  1762.8  5016.2  1763.3
  5032.1 1764.99  5038.5 1767.34  5061.1 1769.29  5110.8 1771.23  5568.8 1779.28
#Mann= 3 ,-1 , 0
  4490.7     .05       0  5006.4     .05       0  5016.2     .05       0
Bank Sta=5006.4,5016.2
XS Rating Curve= 0 ,0
Exp/Cntr=0.3,0.1

Type RM Length L Ch R = 1 ,7548    ,784,784,784
BEGIN DESCRIPTION:
Elm 02 01 7547.86
END DESCRIPTION:
XS GIS Cut Line= 3
      1605079.54      6822339.68      1605555.27      6822586.22
      1606274.03      6822940.39
#Sta/Elev= 30
    4470 1774.15  4701.4  1774.4  4755.9 1774.05  4859.1 1772.11  4872.2  1771.4
  4904.1  1771.1    4933 1769.13  4971.6 1767.26    4983 1766.06  4994.5 1762.66
    4995 1762.16  5003.8 1762.16  5004.3 1762.66  5008.5 1763.03  5016.1 1766.33
    5061 1766.54  5066.6 1767.06  5089.1 1767.02  5105.9  1767.9  5150.4 1768.23
  5184.5 1769.67  5296.8 1769.99  5351.1 1770.94  5373.4 1770.84    5426 1772.25
  5462.6 1772.63  5493.4  1773.6  5605.7 1775.68  5611.2 1776.14  5807.1  1779.4
#Mann= 3 ,-1 , 0
    4470     .05       0  4994.5     .05       0  5004.3     .05       0
Bank Sta=4994.5,5004.3
XS Rating Curve= 0 ,0
Exp/Cntr=0.3,0.1

Type RM Length L Ch R = 1 ,6764    ,1030,1030,1030
BEGIN DESCRIPTION:
Elm 02 01 6763.63
END DESCRIPTION:
XS GIS Cut Line= 3
       1604801.8      6822683.45      1605517.07      6823124.42
       1606050.9      6823370.53
#Sta/Elev= 30
  4160.8  1771.3  4311.9 1770.86  4470.3  1767.5  4601.7 1765.85  4812.2 1767.47
  4848.9 1766.21  4900.9 1765.72  4906.8 1765.05  4937.6 1764.33  4943.5  1763.7
  4958.9  1763.4  4964.8 1761.89  4974.3  1761.9  4975.2 1760.41  4975.7 1759.91
  4984.7 1759.91  4985.2 1760.41  4995.6 1760.99  4999.7 1763.94  5018.4 1765.29
    5024 1767.32  5041.4 1768.95  5046.9 1770.33  5064.4 1770.88  5069.9 1772.57
  5098.3  1772.7  5115.8 1773.89  5184.6 1774.47  5350.8 1777.37  5588.9 1779.66
#Mann= 3 ,-1 , 0
  4160.8     .05       0  4975.2     .05       0  4985.2     .05       0
Bank Sta=4975.2,4985.2
XS Rating Curve= 0 ,0
Exp/Cntr=0.3,0.1

Type RM Length L Ch R = 1 ,5734    ,573,573,573
BEGIN DESCRIPTION:
Elm 02 01 5734.16
END DESCRIPTION:
XS GIS Cut Line= 3
      1604343.45      6822804.97      1604610.82      6823034.14
      1605326.06      6823429.95
#Sta/Elev= 30
  4647.5 1768.68  4977.4 1769.09    4984 1767.57  4991.6 1764.75  4998.2 1761.47
  5004.9 1760.76    5014  1758.7  5022.2 1758.49  5022.7 1757.99  5031.8 1757.99
  5032.3 1758.49  5035.8 1760.07  5050.1 1761.47  5107.3 1762.69  5166.3 1762.11
  5210.1 1763.14  5263.7 1763.37  5328.9 1762.61    5345 1763.19  5372.5 1762.77
  5426.3 1763.51  5541.6 1763.76  5610.2 1765.31  5632.4 1766.68  5654.2 1766.98
  5681.6 1768.65  5735.5  1770.7    5779 1771.45    5793 1772.35  5817.1 1772.27
#Mann= 3 ,-1 , 0
  4647.5     .05       0  5022.2     .05       0  5032.3     .05       0
Bank Sta=5022.2,5032.3
XS Rating Curve= 0 ,0
Exp/Cntr=0.3,0.1

Type RM Length L Ch R = 1 ,5161    ,403,403,403
BEGIN DESCRIPTION:
Elm 02 01 5160.6
END DESCRIPTION:
XS GIS Cut Line= 3
      1604197.66      6823461.22      1604756.65        6823489.
       1605311.1      6823544.44
#Sta/Elev= 30
    4442 1767.32  4609.6 1767.81  4729.7 1766.18  4849.8 1761.42  4929.9 1759.78
    4990 1759.39  5001.7 1757.87  5010.1 1755.22  5015.1 1754.91  5015.6 1754.41
  5024.7 1754.41  5025.2 1754.91  5038.6 1761.26  5043.6 1760.18  5050.3 1761.51
  5070.4 1761.89  5100.5 1761.46  5120.6    1762  5221.1 1761.96  5281.4 1764.44
  5301.5  1766.1  5331.7 1766.89    5340 1767.68  5345.1  1769.1  5351.8  1769.5
  5381.9 1769.62  5412.1 1771.13  5432.2  1770.7  5492.5 1772.68  5558.9  1773.7
#Mann= 3 ,-1 , 0
    4442     .05       0  5015.1     .05       0  5025.2     .05       0
Bank Sta=5015.1,5025.2
XS Rating Curve= 0 ,0
Exp/Cntr=0.3,0.1

Type RM Length L Ch R = 1 ,4758    ,391,391,391
BEGIN DESCRIPTION:
Elm 02 01 4757.66
END DESCRIPTION:
XS GIS Cut Line= 3
      1604352.08      6823761.93      1604701.46      6823874.78
      1605055.21      6824004.99
#Sta/Elev= 30
  4628.6 1764.81  4666.5 1763.88  4698.6 1763.71  4736.8 1762.08  4778.8 1761.31
  4831.9 1759.66  4883.9 1759.03  4890.7 1758.33  4915.4 1757.67  4946.9 1757.51
  4954.8  1756.6  4960.1  1756.8  4967.9 1754.06  4978.5 1754.59    4987 1753.89
  4987.5 1753.39  4996.7 1753.39  4997.2 1753.89  5000.3  1755.3  5010.2 1756.07
  5022.9 1755.65  5042.1 1756.38  5063.5 1759.64  5078.4 1760.89  5084.8 1762.24
  5103.6 1764.43    5134 1765.96    5195 1766.56  5275.7 1768.51  5372.7 1769.31
#Mann= 3 ,-1 , 0
  4628.6     .05       0    4987     .05       0  4997.2     .05       0
Bank Sta=4987,4997.2
XS Rating Curve= 0 ,0
Exp/Cntr=0.3,0.1

Type RM Length L Ch R = 1 ,4367    ,366,366,366
BEGIN DESCRIPTION:
Elm 02 01 4366.83
END DESCRIPTION:
XS GIS Cut Line= 3
      1604141.55      6824022.34      1604536.53      6824204.64
      1605018.27      6824430.32
#Sta/Elev= 30
  4563.8 1763.22  4721.8  1760.8  4735.4 1759.57  4787.9 1759.48  4798.7 1758.36
    4865 1755.81  4941.9 1756.48  4953.1 1754.03    4959 1753.84  4959.5 1753.34
  4968.7 1753.34  4969.2 1753.84  4996.9 1754.86  5030.3 1754.52  5084.6 1758.78
  5112.9 1759.01  5158.6  1760.7  5272.8 1762.71  5278.3 1762.13  5301.1 1762.93
  5323.9 1762.56  5339.5 1761.34  5375.1 1761.52  5392.4 1763.08  5443.6 1764.44
  5460.9 1765.62    5483 1765.62  5505.1 1767.09  5517.6 1766.71  5530.8 1767.34
#Mann= 3 ,-1 , 0
  4563.8     .05       0    4959     .05       0  4969.2     .05       0
Bank Sta=4959,4969.2
XS Rating Curve= 0 ,0
Exp/Cntr=0.3,0.1

Type RM Length L Ch R = 1 ,4001    ,452,452,452
BEGIN DESCRIPTION:
Elm 02 01 4000.98
END DESCRIPTION:
XS GIS Cut Line= 3
      1603875.32      6824340.77      1604292.03      6824450.15
      1604809.39       6824625.5
#Sta/Elev= 30
    4569 1759.52  4651.4 1758.41  4713.4 1759.23  4796.1    1758  4812.9 1756.14
  4928.8 1753.73  4964.1 1749.84  4964.6 1749.34  4974.3 1749.84  4992.6 1751.49
  4998.8 1753.58    5004 1753.58  5008.5  1755.5  5055.8 1754.44  5071.3 1756.21
  5076.9 1759.29  5087.4 1759.27  5097.4  1757.6  5102.7 1759.21  5119.1 1760.76
  5134.1 1758.41  5140.2 1755.86  5150.8 1754.84  5214.1  1753.4  5385.4 1761.57
  5404.2    1761  5411.6 1762.49  5467.6 1763.34  5479.7 1764.83  5546.1 1765.37
#Mann= 3 ,-1 , 0
    4569     .05       0  4964.1     .05       0  4974.3     .05       0
Bank Sta=4964.1,4974.3
XS Rating Curve= 0 ,0
Exp/Cntr=0.3,0.1

Type RM Length L Ch R = 1 ,3549    ,73,73,73
BEGIN DESCRIPTION:
Elm 02 01 3548.96
END DESCRIPTION:
XS GIS Cut Line= 4
      1603967.07      6824518.16      1604230.25      6824775.94
      1604256.29      6824788.09      1604459.46      6824786.35
#Sta/Elev= 30
  4603.8 1759.87  4672.9 1758.87    4687 1759.43  4694.2 1758.13  4715.3 1757.94
  4722.5 1757.14  4771.9  1756.1  4793.2 1755.22  4807.3 1755.56  4814.3 1755.32
  4821.5 1753.59  4828.5 1753.09  4835.6 1751.04  4842.6 1750.78  4849.8 1749.31
  4856.8 1749.18  4879.8 1746.62  4880.3 1746.12  4889.8 1746.12  4890.3 1746.62
  4913.3 1747.01  4955.8 1746.64  5059.6 1746.81  5069.6 1747.52  5089.6 1750.85
  5109.6 1753.54  5129.6 1757.79  5139.6  1759.2  5169.6 1760.81  5204.1 1761.58
#Mann= 3 ,-1 , 0
  4603.8     .05       0  4879.8     .05       0  4890.3     .05       0
Bank Sta=4879.8,4890.3
XS Rating Curve= 0 ,0
Exp/Cntr=0.3,0.1
