--- Elm 02 17.prj (project) ---

Proj Title=Elm 02 17 Base Level Engineering
Current Plan=p01
Default Exp/Contr=0.3,0.1
English Units
Geom File=g01
Flow File=f01
Plan File=p01
BEGIN DESCRIPTION:
Elm 02 17
END DESCRIPTION:

--- Elm 02 17.p01 (plan) ---

Plan Title=Multiple Run
Short Identifier=Multiple
Geom File=g01
Flow File=f01
Subcritical Flow
K Sum by GR= 0
Std Step Tol= 0.01
Critical Tol= 0.01
Num of Std Step Trials= 20
Max Error Tol= 0.3
Flow Tol Ratio= 0.001
Split Flow NTrial= 30
Split Flow Tol= 0.02
Split Flow Ratio= 0.02
Log Output Level= 0
Friction Slope Method= 1
Unsteady Friction Slope Method= 2
Unsteady Bridges Friction Slope Method= 1
Parabolic Critical Depth
Global Vel Dist=  1 , 1 , 1
Global Log Level= 0
CheckData=True
Encroach Param= -1, 0, 0, 0
BEGIN DESCRIPTION:
Multiple Run
END DESCRIPTION:

--- Elm 02 17.f01 (steady flow) ---

Flow Title=Multiple
Number of Profiles=7
Profile Names=10-year,25-year,50-year,1pct_min,100-year,1pct_plu,500-year
River Rch & RM= Elm 02 17,Reach-1,21787
     167     225     272     204     327     450     478
River Rch & RM= Elm 02 17,Reach-1,20739
     305     425     525     401     643     885     979
River Rch & RM= Elm 02 17,Reach-1,12029
     422     598     746     576     922    1270    1430
Boundary for River Rch & Prof#=Elm 02 17,Reach-1,1
Up Type=0
Dn Type=3
Dn Slope=0.001
Boundary for River Rch & Prof#=Elm 02 17,Reach-1,2
Up Type=0
Dn Type=3
Dn Slope=0.001
Boundary for River Rch & Prof#=Elm 02 17,Reach-1,3
Up Type=0
Dn Type=3
Dn Slope=0.001
Boundary for River Rch & Prof#=Elm 02 17,Reach-1,4
Up Type=0
Dn Type=3
Dn Slope=0.001
Boundary for River Rch & Prof#=Elm 02 17,Reach-1,5
Up Type=0
Dn Type=3
Dn Slope=0.001
Boundary for River Rch & Prof#=Elm 02 17,Reach-1,6
Up Type=0
Dn Type=3
Dn Slope=0.001
Boundary for River Rch & Prof#=Elm 02 17,Reach-1,7
Up Type=0
Dn Type=3
Dn Slope=0.001

--- Elm 02 17.g01 (geometry) ---

Geom Title=Existing Conditions

River Reach=Elm 02 17,Reach-1
Reach XY= 30
      1620755.00      6827938.00      1621147.48      6828041.12
      1620397.12      6829694.13      1620021.03      6829920.86
      1620007.77      6830132.64      1619720.64      6830187.58
      1619606.67      6830041.08      1618858.37      6830539.28
      1619255.17      6831317.74      1619146.86      6831694.06
      1618758.04      6832039.42      1618599.59      6833132.83
      1618129.79      6833288.36      1617999.57      6832990.17
      1617348.94      6833096.14      1617108.51      6833296.48
      1616951.18      6833986.42      1616655.07      6834380.73
      1616435.22      6833967.91      1615888.32      6833671.36
      1615453.42      6833091.67      1614266.31      6833490.26
      1613708.67      6834189.59      1613799.54      6834590.45
      1613314.68      6835127.24      1612419.76      6835437.25
      1611961.17      6834745.86      1611506.50      6834791.62
      1610268.61      6835574.76      1609805.00      6836788.00

Type RM Length L Ch R = 1,21787,599,599,599
BEGIN DESCRIPTION:
Elm 02 17 21387.972
END DESCRIPTION:
XS GIS Cut Line= 3
      1620534.16      6828141.28      1620824.98      6827907.40
      1621121.33      6827624.36
#Sta/Elev= 30
  4626.8 1850.18  4658.0 1850.37  4686.8 1849.71  4707.6 1850.09  4771.6 1849.67
  4800.4 1848.62  4857.9 1847.82  4864.3 1847.28  4921.9 1846.79  4935.9 1845.99
  4942.7 1847.05  4949.2 1847.45  4963.5 1847.07  4983.9 1845.74  4984.2 1845.24
  4987.7 1845.24  4987.9 1845.74  4992.3 1846.13  5003.2 1846.13  5006.7 1846.94
  5035.0 1847.89  5098.5 1848.29  5176.5 1849.57  5197.6 1849.19  5254.2 1850.38
  5296.6 1850.46  5318.0 1851.15  5331.9 1850.97  5367.4 1851.76  5409.8 1851.85
#Mann=3,-1,0
  4626.8    0.05       0  4983.9    0.05       0  4987.9    0.05       0
Bank Sta=4983.9,4987.9
Exp/Cntr=0.3,0.1

Type RM Length L Ch R = 1,21188,449,449,449
BEGIN DESCRIPTION:
Elm 02 17 21188.43
END DESCRIPTION:
XS GIS Cut Line= 3
      1620521.12      6828271.52      1621052.35      6828227.25
      1621548.40      6828032.47
#Sta/Elev= 30
  4463.9 1849.29  4558.1 1848.50  4578.2 1847.89  4618.3 1847.85  4758.8 1845.54
  4829.0 1845.64  4889.3 1845.01  4979.6 1845.63  4989.6 1845.35  4995.8 1843.41
  5004.9 1843.03  5005.2 1842.53  5008.7 1842.53  5008.9 1843.03  5042.8 1844.15
  5053.5 1843.95  5128.7 1845.38  5139.5 1844.55  5145.1 1844.81  5161.0 1844.11
  5169.6 1844.13  5174.9 1845.15  5193.2 1844.21  5229.1 1845.94  5278.0 1847.19
  5313.2 1849.00  5332.2 1849.02  5354.4 1849.94  5421.6 1851.34  5529.9 1852.32
#Mann=3,-1,0
  4463.9    0.05       0  5004.9    0.05       0  5008.9    0.05       0
Bank Sta=5004.9,5008.9
Exp/Cntr=0.3,0.1

Type RM Length L Ch R = 1,20739,362,362,362
BEGIN DESCRIPTION:
Elm 02 17 20739.47
END DESCRIPTION:
XS GIS Cut Line= 3
      1620495.09      6828459.03      1620872.66      6828578.81
      1621335.74      6828623.04
#Sta/Elev= 30
  4609.2 1848.21  4682.5 1847.43  4745.5 1845.88  4752.7 1845.04  4777.0 1843.43
  4784.9 1842.36  4797.9 1841.65  4808.4 1841.43  4817.2 1841.91  4829.4 1841.73
  4849.5 1842.29  4887.0 1842.48  4944.8 1843.58  4981.7 1840.28  4982.0 1839.78
  4985.7 1839.78  4986.0 1840.28  4997.3 1840.52  5003.9 1841.36  5037.8 1842.23
  5057.9 1843.53  5067.9 1843.75  5098.1 1843.60  5153.9 1844.26  5218.6 1844.31
  5399.4 1846.91  5429.6 1846.55  5439.6 1847.17  5459.7 1847.03  5470.5 1847.48
#Mann=3,-1,0
  4609.2    0.05       0  4981.7    0.05       0  4986.0    0.05       0
Bank Sta=4981.7,4986
Exp/Cntr=0.3,0.1

Type RM Length L Ch R = 1,20377,341,341,341
BEGIN DESCRIPTION:
Elm 02 17 20377.45
END DESCRIPTION:
XS GIS Cut Line= 3
      1620465.91      6828749.97      1620851.32      6828935.73
      1621260.50      6829036.29
#Sta/Elev= 30
  4571.9 1844.81  4593.1 1844.12  4622.9 1844.16  4628.4 1843.62  4645.5 1843.58
  4659.7 1842.75  4681.9 1843.08  4690.7 1842.41  4781.2 1841.51  4815.1 1839.70
  4892.8 1839.21  4915.0 1839.62  4922.5 1840.74  4928.0 1840.75  4945.1 1839.66
  4973.3 1838.85  4981.6 1838.00  4993.7 1837.64  4994.0 1837.14  4997.8 1837.14
  4998.0 1837.64  4999.0 1838.59  5029.7 1840.01  5044.7 1840.26  5055.0 1840.94
  5065.3 1842.29  5071.3 1842.47  5219.8 1843.51  5237.5 1844.05  5421.1 1844.82
#Mann=3,-1,0
  4571.9    0.05       0  4993.7    0.05       0  4998.0    0.05       0
Bank Sta=4993.7,4998
Exp/Cntr=0.3,0.1

Type RM Length L Ch R = 1,20036,90,90,90
BEGIN DESCRIPTION:
Elm 02 17 20035.92
END DESCRIPTION:
XS GIS Cut Line= 3
      1620204.32      6828992.31      1620605.40      6829155.09
      1620986.88      6829201.96
#Sta/Elev= 30
  4565.6 1840.16  4623.2 1838.08  4647.2 1837.95  4739.0 1838.16  4749.0 1838.50
  4754.4 1838.21  4802.6 1838.37  4814.6 1838.93  4832.1 1838.73  4861.5 1839.96
  4868.5 1839.47  4891.0 1839.62  4900.9 1840.08  4939.2 1840.10  4963.3 1838.90
  4976.4 1836.71  4990.6 1835.93  4990.9 1835.43  4994.7 1835.43  4995.0 1835.93
  5018.2 1836.29  5058.4 1838.05  5098.8 1839.14  5108.9 1839.87  5159.3 1841.14
  5189.5 1841.47  5209.6 1841.17  5260.0 1841.88  5350.7 1842.40  5382.8 1842.24
#Mann=3,-1,0
  4565.6    0.05       0  4990.6    0.05       0  4995.0    0.05       0
Bank Sta=4990.6,4995
Exp/Cntr=0.3,0.1

Type RM Length L Ch R = 1,19946,604,604,604
BEGIN DESCRIPTION:
Elm 02 17 19945.79
END DESCRIPTION:
XS GIS Cut Line= 3
      1620006.43      6829134.25      1620566.34      6829231.91
      1621144.51      6829431.14
#Sta/Elev= 30
  4434.5 1840.95  4463.5 1840.50  4524.4 1837.60  4554.9 1836.77  4601.2 1837.43
  4606.3 1836.74  4625.9 1836.85  4808.6 1838.89  4892.8 1839.05  4910.1 1839.63
  4971.1 1839.12  5009.8 1836.25  5010.1 1835.75  5013.9 1835.75  5014.2 1836.25
  5032.4 1837.11  5037.7 1837.92  5054.3 1838.08  5068.9 1837.55  5094.8 1838.26
  5100.1 1837.92  5162.5 1840.48  5276.5 1841.04  5287.4 1840.02  5313.3 1839.11
  5407.0 1841.67  5432.9 1840.61  5526.5 1840.96  5588.9 1843.58  5614.4 1843.77
#Mann=3,-1,0
  4434.5    0.05       0  5009.8    0.05       0  5014.2    0.05       0
Bank Sta=5009.8,5014.2
Exp/Cntr=0.3,0.1

Type RM Length L Ch R = 1,19342,391,391,391
BEGIN DESCRIPTION:
Elm 02 17 19341.83
END DESCRIPTION:
XS GIS Cut Line= 6
      1619958.31      6829247.56      1620322.85      6829505.35
      1620347.59      6829746.23      1620387.96      6829780.09
      1620481.71      6829764.46      1620796.77      6829892.05
#Sta/Elev= 30
  4313.0 1840.04  4324.9 1838.96  4339.7 1839.07  4411.0 1836.39  4465.8 1835.38
  4466.2 1834.88  4470.2 1834.88  4470.5 1835.38  4512.0 1835.57  4562.5 1837.17
  4740.9 1837.32  4755.7 1840.26  4757.7 1841.58  4812.3 1842.56  4922.9 1842.07
  4973.2 1840.99  4993.4 1839.52  5022.8 1841.08  5061.5 1840.89  5097.2 1842.70
  5102.3 1841.79  5112.2 1841.90  5132.4 1842.88  5148.5 1844.53  5163.7 1844.48
  5170.6 1843.93  5176.0 1842.46  5200.1 1840.58  5347.1 1845.18  5489.3 1852.03
#Mann=3,-1,0
  4313.0    0.05       0  4465.8    0.05       0  4470.5    0.05       0
Bank Sta=4465.8,4470.5
Exp/Cntr=0.3,0.1

Type RM Length L Ch R = 1,18951,913,913,913
BEGIN DESCRIPTION:
Elm 02 17 18951.1
END DESCRIPTION:
XS GIS Cut Line= 3
      1619573.73      6829457.61      1620025.54      6829919.84
      1620383.64      6830182.89
#Sta/Elev= 30
  4356.0 1838.40  4470.3 1837.54  4491.6 1836.52  4505.7 1836.53  4548.1 1834.59
  4555.1 1833.95  4597.6 1832.99  4625.9 1833.12  4654.1 1833.80  4802.7 1834.48
  4873.5 1833.82  4894.6 1834.12  4929.9 1833.46  4958.2 1832.28  4965.3 1832.38
  4970.0 1831.19  4970.3 1830.69  4974.3 1830.69  4974.7 1831.19  4993.6 1831.43
  4998.4 1832.51  5037.1 1832.66  5051.3 1832.00  5064.2 1832.44  5093.5 1832.54
  5108.1 1833.70  5193.8 1835.92  5365.1 1841.65  5400.6 1843.78  5446.7 1845.66
#Mann=3,-1,0
  4356.0    0.05       0  4970.0    0.05       0  4974.7    0.05       0
Bank Sta=4970,4974.7
Exp/Cntr=0.3,0.1

Type RM Length L Ch R = 1,18038,514,514,514
BEGIN DESCRIPTION:
Elm 02 17 18037.57
END DESCRIPTION:
XS GIS Cut Line= 3
      1619245.75      6829760.37      1619512.65      6830134.04
      1619819.94      6830592.36
#Sta/Elev= 30
  4540.7 1834.66  4667.6 1832.42  4753.7 1832.08  4774.6 1831.39  4810.2 1831.52
  4818.8 1831.16  4824.9 1831.64  4845.8 1831.63  4925.7 1829.75  4955.2 1829.74
  4961.3 1830.20  4967.9 1829.96  4976.1 1828.60  4982.2 1828.30  4988.4 1826.72
  4988.8 1826.22  4992.9 1826.22  4993.2 1826.72  4997.0 1826.87  4999.3 1828.34
  5062.9 1829.86  5198.0 1830.47  5279.0 1830.30  5336.0 1831.47  5342.1 1831.94
  5450.1 1832.27  5486.3 1832.82  5501.1 1832.48  5516.1 1833.02  5551.7 1832.78
#Mann=3,-1,0
  4540.7    0.05       0  4988.4    0.05       0  4993.2    0.05       0
Bank Sta=4988.4,4993.2
Exp/Cntr=0.3,0.1

Type RM Length L Ch R = 1,17524,520,520,520
BEGIN DESCRIPTION:
Elm 02 17 17524.24
END DESCRIPTION:
XS GIS Cut Line= 3
      1618796.36      6830026.89      1619115.84      6830280.39
      1619421.57      6830430.67
#Sta/Elev= 30
  4593.6 1835.91  4656.9 1834.30  4706.7 1832.66  4764.3 1831.12  4807.5 1830.65
  4878.0 1828.94  4885.5 1828.98  4892.4 1829.31  4898.8 1828.70  4956.5 1827.65
  4962.9 1827.12  4974.9 1826.90  4975.2 1826.40  4979.4 1826.40  4979.8 1826.90
  4997.7 1827.43  5022.8 1827.28  5029.2 1827.53  5074.1 1827.44  5096.6 1827.73
  5102.2 1827.55  5111.9 1828.02  5124.7 1827.72  5201.1 1828.46  5245.6 1828.62
  5282.0 1829.37  5298.9 1829.50  5304.5 1830.02  5312.5 1829.47  5342.1 1829.94
#Mann=3,-1,0
  4593.6    0.05       0  4974.9    0.03       0  4979.8    0.05       0
Bank Sta=4974.9,4979.8
Exp/Cntr=0.3,0.1

Type RM Length L Ch R = 1,17004,306,306,306
BEGIN DESCRIPTION:
Elm 02 17 17004.18
END DESCRIPTION:
XS GIS Cut Line= 6
      1618462.50      6830590.97      1618726.43      6830679.52
      1618816.71      6830696.88      1618882.68      6830665.63
      1618985.11      6830563.20      1619316.73      6830457.29
#Sta/Elev= 30
  4556.2 1837.30  4752.6 1832.06  4801.4 1829.91  4843.3 1829.80  4855.8 1828.93
  4873.9 1831.15  4902.6 1829.08  4907.7 1830.10  4914.6 1829.12  4926.5 1828.92
  4938.4 1829.25  4955.6 1831.00  4961.2 1830.35  4968.9 1831.80  4978.4 1832.31
  5013.6 1831.90  5070.2 1833.68  5105.6 1832.17  5112.6 1830.86  5119.7 1830.99
  5126.8 1828.65  5133.8 1828.60  5140.8 1826.90  5174.2 1826.07  5238.6 1826.64
  5257.2 1825.77  5257.6 1825.27  5262.2 1825.77  5345.6 1827.77  5492.5 1828.60
#Mann=3,-1,0
  4556.2    0.05       0  5257.2    0.05       0  5262.2    0.05       0
Bank Sta=5257.2,5262.2
Exp/Cntr=0.3,0.1

Type RM Length L Ch R = 1,16698,162,162,162
BEGIN DESCRIPTION:
Elm 02 17 16697.75
END DESCRIPTION:
XS GIS Cut Line= 3
      1618608.86      6830862.64      1619004.69      6830866.55
      1619588.05      6830848.32
#Sta/Elev= 30
  4603.9 1834.76  4637.7 1833.21  4642.7 1833.51  4660.0 1832.34  4680.0 1831.96
  4740.0 1828.71  4800.1 1826.52  4820.1 1825.31  4830.1 1824.12  4860.1 1822.68
  4920.1 1823.12  4940.1 1822.66  4960.1 1824.20  4990.1 1824.51  5002.4 1824.35
  5017.6 1822.04  5017.9 1821.54  5022.2 1821.54  5022.6 1822.04  5040.1 1823.95
  5080.1 1825.08  5180.2 1825.34  5190.2 1824.94  5310.2 1826.26  5350.2 1826.23
  5370.2 1826.71  5390.3 1828.42  5420.3 1829.22  5434.4 1828.89  5583.4 1829.24
#Mann=3,-1,0
  4603.9    0.05       0  5017.6    0.03       0  5022.6    0.05       0
Bank Sta=5017.6,5022.6
Exp/Cntr=0.3,0.1

Type RM Length L Ch R = 1,16536,582,582,582
BEGIN DESCRIPTION:
Elm 02 17 16536.02
END DESCRIPTION:
XS GIS Cut Line= 3
      1618576.92      6831024.10      1619075.00      6831006.74
      1619580.36      6830999.15
#Sta/Elev= 30
  4501.5 1836.52  4569.6 1834.63  4659.7 1831.28  4669.7 1830.34  4699.7 1829.27
  4749.7 1826.55  4759.7 1825.72  4779.7 1822.80  4789.8 1822.19  4839.8 1823.81
  4899.8 1822.67  4929.8 1823.34  4967.4 1822.02  4967.7 1821.52  4972.0 1821.52
  4972.4 1822.02  5009.9 1822.97  5019.9 1822.63  5029.9 1823.64  5039.9 1823.53
  5049.9 1822.60  5069.9 1823.06  5099.9 1822.88  5119.9 1823.58  5269.9 1825.81
  5289.9 1825.56  5309.9 1826.29  5389.9 1827.56  5409.9 1827.30  5505.3 1828.34
#Mann=3,-1,0
  4501.5    0.05       0  4967.4    0.05       0  4972.4    0.05       0
Bank Sta=4967.4,4972.4
Exp/Cntr=0.3,0.1

Type RM Length L Ch R = 1,15954,871,871,871
BEGIN DESCRIPTION:
Elm 02 17 15954.32
END DESCRIPTION:
XS GIS Cut Line= 3
      1618259.52      6831466.57      1619203.95      6831485.66
      1619950.23      6831464.84
#Sta/Elev= 30
  4055.1 1835.84  4140.6 1833.19  4240.6 1829.13  4440.7 1824.31  4530.7 1823.60
  4690.7 1821.02  4800.7 1821.30  4860.7 1820.44  4930.8 1821.37  4940.8 1821.17
  4960.8 1819.75  4978.2 1819.35  4978.6 1818.85  4983.0 1818.85  4983.4 1819.35
  4997.8 1820.58  5020.8 1820.90  5040.8 1821.97  5070.8 1822.08  5080.8 1822.77
  5090.5 1822.25  5095.5 1822.77  5130.8 1823.96  5210.9 1824.92  5350.9 1828.14
  5461.0 1830.07  5481.0 1830.87  5601.0 1833.02  5711.1 1835.82  5746.3 1836.16
#Mann=3,-1,0
  4055.1    0.05       0  4978.2    0.05       0  4983.4    0.05       0
Bank Sta=4978.2,4983.4
Exp/Cntr=0.3,0.1

Type RM Length L Ch R = 1,15083,91,91,91
BEGIN DESCRIPTION:
Elm 02 17 15082.64
END DESCRIPTION:
XS GIS Cut Line= 6
      1618181.00      6832117.49      1618644.57      6832141.80
      1618804.30      6832141.80      1618873.74      6832077.56
      1619007.42      6831877.91      1619361.63      6831727.59
#Sta/Elev= 30
  4379.4 1827.36  4523.6 1825.51  4677.2 1821.74  4794.0 1817.80  4841.3 1815.05
  4864.0 1815.82  4884.0 1818.21  4894.0 1818.67  4924.0 1812.57  4934.0 1811.73
  4998.5 1811.60  4998.9 1811.10  5003.8 1811.60  5063.0 1811.97  5100.7 1813.14
  5121.3 1816.62  5127.3 1818.56  5148.3 1816.23  5301.4 1819.35  5351.3 1819.70
  5398.6 1823.35  5404.1 1823.17  5411.6 1824.30  5422.3 1823.62  5427.7 1824.50
  5433.3 1823.22  5498.5 1824.13  5504.2 1823.50  5556.9 1824.79  5723.0 1826.93
#Mann=3,-1,0
  4379.4    0.05       0  4998.5    0.05       0  5003.8    0.05       0
Bank Sta=4998.5,5003.8
Exp/Cntr=0.3,0.1

Type RM Length L Ch R = 1,14992,82,82,82
BEGIN DESCRIPTION:
Elm 02 17 14991.57
END DESCRIPTION:
XS GIS Cut Line= 6
      1618172.34      6832204.30      1618535.20      6832244.23
      1618701.87      6832244.23      1618882.42      6832209.51
      1619010.89      6831968.19      1619398.02      6831802.27
#Sta/Elev= 30
  4365.3 1825.73  4689.9 1820.14  4722.1 1824.36  4830.1 1822.43  4930.4 1825.35
  5042.5 1825.60  5068.9 1822.66  5074.1 1824.64  5098.5 1825.36  5114.1 1821.10
  5119.9 1823.68  5129.6 1821.02  5135.5 1824.30  5151.0 1821.40  5156.8 1824.97
  5172.4 1822.37  5178.2 1825.34  5187.9 1823.89  5245.3 1824.24  5260.0 1822.22
  5277.4 1823.96  5282.9 1821.82  5300.3 1823.82  5305.8 1821.31  5344.5 1823.25
  5387.8 1818.98  5388.2 1818.48  5393.1 1818.98  5588.3 1824.43  5776.5 1826.99
#Mann=3,-1,0
  4365.3    0.05       0  5387.8    0.05       0  5393.1    0.05       0
Bank Sta=5387.8,5393.1
Exp/Cntr=0.3,0.1

Type RM Length L Ch R = 1,14910,370,370,370
BEGIN DESCRIPTION:
Elm 02 17 14909.79
END DESCRIPTION:
XS GIS Cut Line= 6
      1618115.09      6832259.86      1618611.59      6832308.47
      1618788.67      6832308.47      1618941.45      6832282.42
      1619054.30      6832082.77      1619436.20      6831921.33
#Sta/Elev= 30
  4327.7 1824.70  4759.7 1820.03  4767.6 1822.04  4772.6 1821.36  4779.8 1822.38
  4789.8 1820.26  4860.0 1818.33  4920.0 1814.94  4950.0 1814.50  4960.0 1813.76
  5003.7 1814.48  5020.2 1813.07  5033.2 1812.87  5033.6 1812.37  5038.1 1812.37
  5038.5 1812.87  5050.6 1813.17  5090.9 1816.67  5101.4 1816.91  5141.9 1817.49
  5178.5 1817.10  5209.7 1818.02  5237.7 1817.60  5324.5 1819.03  5491.0 1820.40
  5567.5 1821.77  5638.4 1823.97  5649.5 1823.55  5703.6 1825.47  5802.6 1827.33
#Mann=3,-1,0
  4327.7    0.05       0  5033.2    0.05       0  5038.5    0.05       0
Bank Sta=5033.2,5038.5
Exp/Cntr=0.3,0.1

Type RM Length L Ch R = 1,14540,508,508,508
BEGIN DESCRIPTION:
Elm 02 17 14539.66
END DESCRIPTION:
XS GIS Cut Line= 3
      1618196.42      6832525.28      1618705.08      6832653.75
      1619201.66      6832778.33
#Sta/Elev= 30
  4476.0 1817.64  4545.0 1817.63  4591.2 1817.14  4750.2 1816.61  4796.4 1816.01
  4887.1 1815.78  4938.7 1814.58  4969.6 1813.08  4996.4 1811.18  4996.8 1810.68
  5001.4 1810.68  5001.8 1811.18  5010.9 1811.62  5084.0 1811.90  5103.6 1812.63
  5155.2 1813.49  5161.1 1813.86  5166.3 1813.62  5202.3 1814.37  5237.7 1814.08
  5243.5 1813.32  5248.6 1813.76  5299.5 1814.08  5325.8 1815.98  5351.1 1815.83
  5423.2 1817.53  5443.9 1818.70  5474.8 1821.09  5505.7 1822.62  5512.6 1823.33
#Mann=3,-1,0
  4476.0    0.05       0  4996.4    0.05       0  5001.8    0.05       0
Bank Sta=4996.4,5001.8
Exp/Cntr=0.3,0.1

Type RM Length L Ch R = 1,14032,502,502,502
BEGIN DESCRIPTION:
Elm 02 17 14032.44
END DESCRIPTION:
XS GIS Cut Line= 3
      1618146.07      6832580.85      1618602.65      6833132.92
      1618830.03      6833339.47
#Sta/Elev= 30
  4287.3 1816.40  4448.1 1813.84  4497.6 1813.94  4511.9 1814.82  4518.4 1814.60
  4526.3 1812.81  4532.7 1813.85  4540.6 1812.41  4547.1 1812.94  4554.9 1812.20
  4575.7 1812.84  4724.8 1811.19  4859.7 1810.79  4894.9 1809.09  4902.7 1809.18
  4923.5 1812.63  4937.9 1810.36  4984.6 1808.22  4985.1 1807.72  4990.1 1808.22
  5001.6 1810.05  5016.2 1810.87  5058.7 1811.54  5087.1 1813.89  5122.3 1814.27
  5221.6 1820.76  5228.4 1822.35  5256.7 1824.78  5306.1 1827.10  5310.9 1828.10
#Mann=3,-1,0
  4287.3    0.05       0  4984.6    0.05       0  4990.1    0.05       0
Bank Sta=4984.6,4990.1
Exp/Cntr=0.3,0.1

Type RM Length L Ch R = 1,13530,402,402,402
BEGIN DESCRIPTION:
Elm 02 17 13530.39
END DESCRIPTION:
XS GIS Cut Line= 3
      1618213.93      6832833.24      1618183.55      6833288.07
      1618176.61      6833429.56
#Sta/Elev= 30
  4544.0 1811.21  4603.4 1810.19  4649.0 1808.80  4689.1 1807.19  4699.1 1806.58
  4706.4 1806.50  4706.8 1806.00  4711.5 1806.00  4711.9 1806.50  4719.1 1807.06
  4739.2 1809.66  4748.6 1809.14  4753.6 1809.87  4769.3 1808.26  4829.4 1808.29
  4879.5 1808.72  4903.8 1809.27  4919.6 1808.98  4939.6 1809.10  4949.7 1808.80
  4959.7 1808.94  4969.7 1808.63  4989.7 1806.72  5002.3 1806.78  5009.8 1808.25
  5029.8 1811.38  5049.8 1812.62  5068.6 1813.26  5119.9 1814.39  5141.5 1814.45
#Mann=3,-1,0
  4544.0    0.05       0  4706.4    0.05       0  4711.9    0.05       0
Bank Sta=4706.4,4711.9
Exp/Cntr=0.3,0.1

Type RM Length L Ch R = 1,13128,307,307,307
BEGIN DESCRIPTION:
Elm 02 17 13128.05
END DESCRIPTION:
XS GIS Cut Line= 3
      1618163.59      6832799.34      1618038.58      6833023.31
      1617897.06      6833304.63
#Sta/Elev= 30
  4745.3 1811.50  4794.5 1809.67  4846.8 1809.41  4853.9 1808.93  4869.7 1808.37
  4875.6 1807.80  4904.1 1806.81  4927.0 1806.34  4935.0 1806.59  4940.8 1806.27
  4949.9 1806.19  4956.7 1805.76  4991.6 1805.18  4992.1 1804.68  4996.8 1804.68
  4997.2 1805.18  5000.2 1805.52  5007.2 1805.64  5029.4 1807.06  5051.8 1806.89
  5067.0 1807.15  5074.2 1806.98  5083.7 1807.24  5089.3 1807.05  5128.4 1807.32
  5178.6 1807.18  5240.0 1808.23  5245.6 1808.10  5275.7 1808.44  5316.7 1809.16
#Mann=3,-1,0
  4745.3    0.05       0  4991.6    0.05       0  4997.2    0.05       0
Bank Sta=4991.6,4997.2
Exp/Cntr=0.3,0.1

Type RM Length L Ch R = 1,12821,452,452,452
BEGIN DESCRIPTION:
Elm 02 17 12820.67
END DESCRIPTION:
XS GIS Cut Line= 3
      1617745.34      6832758.43      1617743.60      6832991.08
      1617743.60      6833348.73
#Sta/Elev= 30
  4769.4 1809.30  4789.0 1808.87  4799.0 1808.35  4809.0 1808.21  4819.0 1808.20
  4839.0 1808.85  4869.0 1808.73  4919.0 1807.61  4939.0 1805.88  4949.0 1804.65
  4959.0 1804.00  4979.0 1803.20  4989.0 1803.21  4998.0 1803.55  5019.0 1803.39
  5039.0 1804.08  5069.0 1804.45  5109.0 1804.14  5129.0 1803.65  5146.2 1802.94
  5146.6 1802.44  5151.3 1802.44  5151.8 1802.94  5159.0 1803.57  5169.0 1803.91
  5209.0 1804.92  5219.0 1805.40  5269.0 1806.80  5299.0 1807.33  5359.7 1807.60
#Mann=3,-1,0
  4769.4    0.05       0  5146.2    0.05       0  5151.8    0.05       0
Bank Sta=5146.2,5151.8
Exp/Cntr=0.3,0.1

Type RM Length L Ch R = 1,12369,340,340,340
BEGIN DESCRIPTION:
Elm 02 17 12368.95
END DESCRIPTION:
XS GIS Cut Line= 3
      1617106.43      6832869.53      1617332.15      6833114.34
      1617597.59      6833423.15
#Sta/Elev= 30
  4668.2 1813.63  4708.3 1813.61  4779.2 1809.83  4878.5 1803.39  4885.3 1801.40
  4892.7 1801.31  4899.5 1800.19  4935.2 1801.24  4942.0 1801.89  4956.2 1801.19
  4963.5 1799.59  5019.5 1801.18  5048.0 1800.23  5076.6 1800.27  5090.8 1801.00
  5126.0 1801.00  5140.2 1800.78  5162.2 1798.91  5173.6 1798.73  5174.1 1798.23
  5178.8 1798.23  5179.2 1798.73  5190.6 1799.42  5197.3 1801.01  5203.9 1801.83
  5260.9 1804.20  5332.2 1804.13  5367.4 1804.57  5395.9 1803.91  5408.4 1804.49
#Mann=3,-1,0
  4668.2    0.05       0  5173.6    0.05       0  5179.2    0.05       0
Bank Sta=5173.6,5179.2
Exp/Cntr=0.3,0.1

Type RM Length L Ch R = 1,12029,840,840,840
BEGIN DESCRIPTION:
Elm 02 17 12029.24
END DESCRIPTION:
XS GIS Cut Line= 3
      1616924.18      6833213.31      1617099.51      6833341.77
      1617400.82      6833627.50
#Sta/Elev= 30
  4784.5 1810.33  4810.3 1810.39  4852.7 1809.76  4902.9 1807.91  4923.7 1806.30
  4932.2 1805.15  4938.4 1804.96  4959.2 1801.89  4982.3 1797.66  4988.5 1796.82
  5001.9 1796.96  5014.1 1796.55  5014.6 1796.05  5019.8 1796.05  5020.3 1796.55
  5024.1 1797.53  5038.3 1798.96  5073.9 1800.02  5088.0 1799.64  5094.9 1799.10
  5109.1 1797.00  5187.1 1798.53  5201.3 1799.13  5222.3 1800.55  5229.6 1800.36
  5236.5 1800.82  5250.6 1800.87  5328.3 1803.10  5356.6 1803.30  5417.1 1804.56
#Mann=3,-1,0
  4784.5    0.05       0  5014.1    0.05       0  5020.3    0.05       0
Bank Sta=5014.1,5020.3
Exp/Cntr=0.3,0.1

Type RM Length L Ch R = 1,11189,254,254,254
BEGIN DESCRIPTION:
Elm 02 17 11189.09
END DESCRIPTION:
XS GIS Cut Line= 3
      1616907.38      6833495.58      1616879.60      6834117.06
      1616900.43      6834643.05
#Sta/Elev= 30
  4382.5 1805.89  4465.0 1803.34  4543.9 1801.59  4575.1 1801.34  4635.2 1799.84
  4745.3 1798.54  4771.0 1798.35  4795.3 1798.79  4815.3 1798.41  4835.4 1797.50
  4855.4 1797.36  4875.4 1796.57  4905.4 1796.14  4915.4 1795.28  4955.5 1794.25
  4998.1 1794.27  4999.5 1793.55  5000.0 1793.05  5005.2 1793.05  5005.7 1793.55
  5025.6 1794.32  5045.6 1795.78  5065.6 1796.31  5095.6 1796.14  5135.6 1796.61
  5175.7 1796.16  5195.7 1796.40  5255.7 1796.17  5325.8 1796.92  5531.0 1804.01
#Mann=3,-1,0
  4382.5    0.05       0  4999.5    0.03       0  5005.7    0.05       0
Bank Sta=4999.5,5005.7
Exp/Cntr=0.3,0.1

Type RM Length L Ch R = 1,10935,504,504,504
BEGIN DESCRIPTION:
Elm 02 17 10935.17
END DESCRIPTION:
XS GIS Cut Line= 3
      1616718.14      6833492.07      1616732.03      6834316.71
      1616744.18      6834618.81
#Sta/Elev= 30
  4181.6 1805.57  4267.5 1802.90  4292.2 1802.52  4337.6 1801.19  4357.6 1800.88
  4427.6 1799.05  4467.6 1798.59  4517.6 1797.40  4607.6 1796.10  4677.6 1795.59
  4817.6 1795.72  4867.6 1795.57  4897.6 1794.84  4917.6 1794.89  4957.6 1794.38
  4977.6 1793.09  4994.5 1792.34  4995.0 1791.84  5000.3 1791.84  5000.8 1792.34
  5004.5 1792.80  5017.7 1792.85  5037.7 1793.62  5057.7 1794.98  5067.7 1794.99
  5167.8 1797.18  5203.7 1798.43  5208.7 1798.29  5277.9 1801.02  5308.7 1801.85
#Mann=3,-1,0
  4181.6    0.05       0  4994.5    0.05       0  5000.8    0.05       0
Bank Sta=4994.5,5000.8
Exp/Cntr=0.3,0.1

Type RM Length L Ch R = 1,10431,290,290,290
BEGIN DESCRIPTION:
Elm 02 17 10430.74
END DESCRIPTION:
XS GIS Cut Line= 3
      1616590.98      6833707.33      1616480.29      6834069.35
      1616393.06      6834350.56
#Sta/Elev= 30
  4626.9 1798.61  4669.6 1796.90  4729.9 1795.39  4735.1 1794.91  4762.7 1794.76
  4826.3 1792.81  4833.5 1792.87  4838.7 1792.42  4857.7 1793.30  4866.3 1793.22
  4899.1 1792.15  4909.9 1791.41  4930.9 1791.50  4942.3 1790.52  4969.9 1790.28
  4990.4 1789.66  4990.9 1789.16  4996.3 1789.16  4996.8 1789.66  5005.5 1790.14
  5007.9 1791.93  5040.5 1793.09  5078.3 1792.67  5105.6 1793.02  5119.2 1792.57
  5150.6 1792.92  5176.0 1792.79  5223.9 1793.57  5255.3 1795.13  5299.9 1795.41
#Mann=3,-1,0
  4626.9    0.05       0  4990.4    0.05       0  4996.8    0.05       0
Bank Sta=4990.4,4996.8
Exp/Cntr=0.3,0.1

Type RM Length L Ch R = 1,10141,236,236,236
BEGIN DESCRIPTION:
Elm 02 17 10141.45
END DESCRIPTION:
XS GIS Cut Line= 3
      1616445.28      6833613.37      1616305.33      6833845.55
      1616166.04      6834084.17
#Sta/Elev= 30
  4731.1 1800.76  4736.2 1800.76  4757.4 1799.36  4778.7 1797.48  4815.6 1795.04
  4837.0 1793.16  4879.7 1791.70  4901.1 1791.30  4923.3 1791.58  4932.1 1791.16
  4937.9 1791.36  4946.7 1791.17  4959.3 1791.63  4974.8 1791.68  4996.2 1790.30
  5000.7 1789.20  5006.5 1789.20  5014.4 1788.39  5014.9 1787.89  5020.3 1787.89
  5020.8 1788.39  5062.9 1789.33  5097.8 1791.23  5120.8 1791.85  5129.2 1792.63
  5144.0 1793.14  5215.2 1793.29  5230.9 1793.63  5236.7 1793.41  5278.5 1793.51
#Mann=3,-1,0
  4731.1    0.05       0  5014.4    0.05       0  5020.8    0.05       0
Bank Sta=5014.4,5020.8
Exp/Cntr=0.3,0.1

Type RM Length L Ch R = 1,9905,340,340,340
BEGIN DESCRIPTION:
Elm 02 17 9904.66
END DESCRIPTION:
XS GIS Cut Line= 3
      1616500.85      6833304.91      1616098.30      6833743.26
      1615959.18      6834036.60
#Sta/Elev= 30
  4407.7 1801.95  4506.3 1799.26  4527.3 1797.56  4541.4 1798.41  4590.8 1794.79
  4612.3 1794.62  4619.1 1793.33  4626.5 1793.97  4661.7 1791.34  4669.1 1792.10
  4675.9 1790.53  4683.3 1791.39  4690.0 1789.92  4704.2 1791.67  4711.0 1790.10
  4718.4 1791.23  4725.2 1790.18  4732.6 1791.29  4739.4 1789.96  4760.9 1791.15
  4796.1 1789.76  4852.8 1790.07  4888.0 1788.94  4937.9 1791.05  5001.4 1788.43
  5043.0 1788.18  5043.5 1787.68  5049.4 1788.18  5119.9 1792.01  5327.5 1792.78
#Mann=3,-1,0
  4407.7    0.05       0  5043.0    0.05       0  5049.4    0.05       0
Bank Sta=5043,5049.4
Exp/Cntr=0.3,0.1

Type RM Length L Ch R = 1,9565,479,479,479
BEGIN DESCRIPTION:
Elm 02 17 9565.18
END DESCRIPTION:
XS GIS Cut Line= 3
      1615990.89      6833142.11      1615811.84      6833596.78
      1615712.19      6834013.78
#Sta/Elev= 30
  4513.8 1801.79  4539.9 1800.95  4569.6 1798.24  4594.0 1797.24  4623.8 1794.98
  4638.4 1793.66  4659.8 1790.26  4678.0 1789.28  4692.1 1786.76  4704.5 1785.87
  4705.0 1785.37  4710.4 1785.37  4710.9 1785.87  4713.6 1786.46  4732.1 1786.86
  4745.8 1786.17  4761.9 1786.59  4767.3 1787.81  4786.3 1788.26  4853.3 1789.15
  4917.8 1789.03  4948.8 1788.34  4993.0 1786.32  5005.7 1786.43  5009.6 1787.94
  5034.6 1788.66  5056.8 1790.26  5116.8 1790.99  5267.2 1791.67  5431.2 1791.25
#Mann=3,-1,0
  4513.8    0.05       0  4704.5    0.05       0  4710.9    0.05       0
Bank Sta=4704.5,4710.9
Exp/Cntr=0.3,0.1

Type RM Length L Ch R = 1,9086,606,606,606
BEGIN DESCRIPTION:
Elm 02 17 9085.92
END DESCRIPTION:
XS GIS Cut Line= 3
      1615674.41      6832940.96      1615624.93      6833189.66
      1615602.84      6833834.21
#Sta/Elev= 30
  4749.8 1801.24  4767.2 1800.64  4777.4 1799.64  4787.6 1800.39  4797.8 1798.98
  4818.2 1798.22  4838.5 1796.83  4858.9 1796.26  4925.7 1791.65  4950.7 1788.72
  4960.9 1788.60  4971.1 1786.76  4976.8 1783.94  4988.0 1783.63  4988.5 1783.13
  4994.4 1783.13  4994.9 1783.63  5000.0 1784.30  5011.7 1784.79  5021.7 1786.12
  5051.7 1786.83  5131.8 1787.35  5147.1 1786.38  5152.1 1787.21  5241.9 1787.38
  5271.9 1787.85  5281.9 1788.52  5371.9 1789.44  5391.9 1789.10  5648.3 1789.86
#Mann=3,-1,0
  4749.8    0.05       0  4988.0    0.05       0  4994.9    0.05       0
Bank Sta=4988,4994.9
Exp/Cntr=0.3,0.1

Type RM Length L Ch R = 1,8480,242,242,242
BEGIN DESCRIPTION:
Elm 02 17 8479.92
END DESCRIPTION:
XS GIS Cut Line= 6
      1615012.26      6832810.92      1615086.49      6833210.69
      1615117.74      6833252.36      1615189.35      6833253.66
      1615249.25      6833209.39      1615536.54      6833783.98
#Sta/Elev= 30
  4596.2 1793.20  4836.8 1790.51  4874.2 1788.62  4887.6 1789.20  4925.3 1786.33
  4930.4 1788.08  4968.7 1785.75  4973.8 1787.33  5007.3 1784.69  5013.5 1787.20
  5021.8 1786.73  5028.1 1788.23  5062.2 1788.55  5088.7 1785.91  5093.7 1788.44
  5102.3 1789.13  5126.6 1787.58  5133.8 1788.80  5170.9 1788.79  5177.7 1787.69
  5201.1 1789.20  5220.7 1784.03  5271.0 1784.30  5300.2 1783.06  5306.7 1780.78
  5307.2 1780.28  5313.7 1780.78  5322.5 1782.95  5444.3 1787.36  5843.5 1789.10
#Mann=3,-1,0
  4596.2    0.05       0  5306.7    0.05       0  5313.7    0.05       0
Bank Sta=5306.7,5313.7
Exp/Cntr=0.3,0.1

Type RM Length L Ch R = 1,8238,316,316,316
BEGIN DESCRIPTION:
Elm 02 17 8237.84
END DESCRIPTION:
XS GIS Cut Line= 3
      1614839.78      6832996.38      1614881.45      6833311.46
      1614869.73      6833819.30
#Sta/Elev= 30
  4682.2 1788.32  4754.4 1787.40  4759.8 1786.82  4764.9 1787.29  4774.6 1786.29
  4804.9 1785.60  4895.7 1785.77  4946.1 1785.19  4956.2 1783.67  4985.2 1781.61
  4995.8 1780.25  5006.6 1779.74  5036.6 1779.52  5046.6 1780.14  5056.6 1781.30
  5062.2 1781.22  5076.6 1779.84  5106.6 1780.39  5136.6 1780.08  5153.1 1779.22
  5153.6 1778.72  5159.6 1778.72  5160.1 1779.22  5176.6 1780.00  5196.6 1780.15
  5206.6 1781.69  5266.6 1783.47  5306.6 1784.03  5346.7 1785.40  5508.0 1789.03
#Mann=3,-1,0
  4682.2    0.05       0  5153.1    0.05       0  5160.1    0.05       0
Bank Sta=5153.1,5160.1
Exp/Cntr=0.3,0.1

Type RM Length L Ch R = 1,7922,271,271,271
BEGIN DESCRIPTION:
Elm 02 17 7921.52
END DESCRIPTION:
XS GIS Cut Line= 3
      1614555.93      6833144.80      1614594.99      6833392.19
      1614645.66      6833763.79
#Sta/Elev= 30
  4752.8 1787.33  4816.8 1786.50  4910.1 1784.36  4928.1 1783.36  4938.3 1782.46
  4948.4 1780.91  4958.5 1780.43  4967.4 1778.56  4972.5 1778.46  4978.8 1779.00
  4995.1 1778.36  4995.6 1777.86  5001.7 1777.86  5002.2 1778.36  5019.2 1779.11
  5029.3 1780.49  5037.3 1781.10  5059.6 1781.55  5069.7 1781.32  5109.7 1781.56
  5120.1 1781.93  5160.5 1782.21  5170.6 1781.67  5192.1 1781.41  5200.9 1781.74
  5211.0 1781.11  5259.4 1781.06  5264.4 1781.34  5331.7 1782.06  5378.3 1783.66
#Mann=3,-1,0
  4752.8    0.05       0  4995.1    0.05       0  5002.2    0.05       0
Bank Sta=4995.1,5002.2
Exp/Cntr=0.3,0.1

Type RM Length L Ch R = 1,7651,241,241,241
BEGIN DESCRIPTION:
Elm 02 17 7651.22
END DESCRIPTION:
XS GIS Cut Line= 3
      1614224.60      6833283.74      1614355.13      6833485.09
      1614584.31      6833782.33
#Sta/Elev= 30
  4761.9 1788.05  4787.5 1787.42  4808.6 1787.28  4823.8 1786.52  4829.8 1786.74
  4850.9 1785.91  4896.3 1784.98  4923.4 1783.58  4945.7 1780.81  4953.7 1779.21
  4959.6 1778.68  4971.2 1775.68  4971.7 1775.18  4977.9 1775.18  4978.4 1775.68
  4981.5 1777.02  4995.9 1778.13  5000.6 1778.84  5046.2 1780.04  5054.4 1779.94
  5075.2 1780.55  5096.0 1780.54  5110.5 1780.90  5154.0 1780.19  5160.3 1780.73
  5168.5 1780.22  5210.1 1780.12  5232.8 1779.42  5318.0 1781.40  5377.2 1783.41
#Mann=3,-1,0
  4761.9    0.05       0  4971.2    0.05       0  4978.4    0.05       0
Bank Sta=4971.2,4978.4
Exp/Cntr=0.3,0.1

Type RM Length L Ch R = 1,7410,326,326,326
BEGIN DESCRIPTION:
Elm 02 17 7409.65
END DESCRIPTION:
XS GIS Cut Line= 3
      1614007.25      6833419.17      1614158.60      6833583.02
      1614420.58      6833860.95
#Sta/Elev= 30
  4778.4 1786.46  4860.7 1784.90  4889.1 1783.78  4903.2 1783.02  4910.6 1781.57
  4924.8 1780.27  4931.6 1780.13  4939.0 1778.91  4945.8 1779.45  4953.1 1777.87
  4977.4 1776.07  4977.9 1775.57  4984.1 1775.57  4984.6 1776.07  4995.1 1777.99
  5001.4 1778.23  5037.7 1777.46  5066.0 1778.87  5101.6 1778.61  5129.9 1779.28
  5144.1 1779.20  5172.4 1777.80  5186.6 1777.33  5193.4 1777.62  5200.7 1777.06
  5214.5 1777.43  5235.9 1779.10  5271.1 1779.69  5341.9 1781.84  5383.4 1782.16
#Mann=3,-1,0
  4778.4    0.05       0  4977.4    0.05       0  4984.6    0.05       0
Bank Sta=4977.4,4984.6
Exp/Cntr=0.3,0.1

Type RM Length L Ch R = 1,7084,302,302,302
BEGIN DESCRIPTION:
Elm 02 17 7083.76
END DESCRIPTION:
XS GIS Cut Line= 4
      1613901.75      6833608.69      1614053.86      6833760.80
      1614147.61      6833789.97      1614432.88      6833893.58
#Sta/Elev= 30
  4687.1 1783.00  4710.1 1782.46  4717.2 1782.61  4724.3 1781.99  4759.6 1780.52
  4837.4 1778.96  4851.5 1779.01  4858.6 1778.50  4872.8 1778.66  4905.4 1777.70
  4909.1 1777.32  4987.2 1776.25  4996.4 1774.68  5007.8 1774.39  5008.3 1773.89
  5014.5 1773.89  5015.0 1774.39  5018.9 1776.34  5029.5 1777.28  5042.0 1777.92
  5067.3 1778.25  5092.6 1778.91  5104.0 1779.52  5123.2 1779.68  5128.5 1780.03
  5178.5 1781.00  5215.0 1781.33  5240.3 1781.96  5284.9 1782.07  5303.9 1782.77
#Mann=3,-1,0
  4687.1    0.05       0  5007.8    0.05       0  5015.0    0.05       0
Bank Sta=5007.8,5015
Exp/Cntr=0.3,0.1

Type RM Length L Ch R = 1,6782,93,93,93
BEGIN DESCRIPTION:
Elm 02 17 6782.45
END DESCRIPTION:
XS GIS Cut Line= 4
      1613866.64      6833645.53      1613898.76      6833878.17
      1613918.73      6833974.53      1614156.54      6834206.27
#Sta/Elev= 30
  4668.4 1782.58  4711.3 1780.88  4731.5 1780.61  4771.8 1779.13  4822.3 1778.46
  4838.3 1777.74  4905.7 1776.09  4913.9 1775.56  4933.7 1775.64  4943.9 1775.28
  4958.9 1775.56  4974.6 1774.92  4984.8 1773.76  4997.3 1773.00  4997.8 1772.50
  5004.0 1772.50  5004.5 1773.00  5008.6 1774.00  5022.8 1775.16  5029.7 1775.39
  5036.9 1776.19  5051.0 1776.58  5065.2 1776.75  5072.2 1776.50  5142.9 1777.86
  5178.2 1778.13  5185.3 1778.49  5220.6 1778.23  5241.9 1778.67  5333.7 1778.87
#Mann=3,-1,0
  4668.4    0.05       0  4997.3    0.05       0  5004.5    0.05       0
Bank Sta=4997.3,5004.5
Exp/Cntr=0.3,0.1

Type RM Length L Ch R = 1,6689,228,228,228
BEGIN DESCRIPTION:
Elm 02 17 6688.89
END DESCRIPTION:
XS GIS Cut Line= 5
      1613682.62      6833697.63      1613777.23      6833894.67
      1613835.39      6834010.12      1613869.25      6834096.92
      1614089.76      6834217.60
#Sta/Elev= 30
  4654.0 1785.55  4687.7 1784.86  4699.2 1783.93  4709.9 1783.63  4721.9 1783.84
  4739.0 1783.12  4744.5 1783.62  4767.2 1781.41  4789.8 1777.49  4806.9 1776.78
  4829.6 1776.36  4852.2 1776.46  4897.0 1777.71  4932.3 1777.61  4947.3 1774.75
  4951.1 1773.63  4951.6 1773.13  4957.8 1773.13  4958.3 1773.63  4977.1 1774.55
  5015.1 1774.87  5069.5 1776.04  5092.9 1775.68  5145.4 1775.96  5151.1 1775.72
  5204.2 1776.71  5210.9 1777.14  5261.2 1777.83  5270.6 1777.51  5346.4 1778.24
#Mann=3,-1,0
  4654.0    0.05       0  4951.1    0.05       0  4958.3    0.05       0
Bank Sta=4951.1,4958.3
Exp/Cntr=0.3,0.1

Type RM Length L Ch R = 1,6461,445,445,445
BEGIN DESCRIPTION:
Elm 02 17 6461.17
END DESCRIPTION:
XS GIS Cut Line= 3
      1613208.05      6834157.12      1613710.70      6834190.98
      1614141.52      6834236.40
#Sta/Elev= 30
  4498.5 1782.19  4525.5 1781.47  4575.6 1780.92  4645.8 1778.88  4715.9 1777.79
  4746.0 1775.84  4786.1 1774.84  4806.1 1774.75  4856.3 1775.50  4896.3 1775.17
  4966.5 1775.36  4976.5 1773.48  4983.0 1771.07  4983.5 1770.57  4989.7 1770.57
  4990.2 1771.07  4996.6 1772.10  5001.9 1773.58  5026.7 1774.21  5107.2 1774.85
  5114.6 1775.28  5119.6 1774.87  5137.3 1774.41  5187.6 1776.12  5217.8 1776.73
  5288.2 1777.21  5305.5 1777.74  5328.4 1777.54  5358.6 1778.11  5435.5 1778.56
#Mann=3,-1,0
  4498.5    0.05       0  4983.0    0.05       0  4990.2    0.05       0
Bank Sta=4983,4990.2
Exp/Cntr=0.3,0.1

Type RM Length L Ch R = 1,6016,453,453,453
BEGIN DESCRIPTION:
Elm 02 17 6015.54
END DESCRIPTION:
XS GIS Cut Line= 3
      1613066.18      6834585.51      1613805.75      6834579.00
      1614209.37      6834633.68
#Sta/Elev= 30
  4262.7 1779.96  4371.5 1779.46  4391.5 1778.66  4451.5 1775.19  4481.5 1774.09
  4547.1 1772.58  4701.5 1771.61  4741.5 1772.58  4791.5 1772.86  4881.5 1772.47
  4901.5 1771.87  4941.5 1772.77  4951.5 1772.65  4987.7 1770.96  4988.2 1770.46
  4994.8 1770.46  4995.3 1770.96  5011.6 1771.32  5029.4 1773.95  5034.5 1773.67
  5041.9 1774.38  5052.0 1774.71  5213.5 1776.08  5223.5 1775.83  5263.9 1776.49
  5284.1 1775.85  5329.8 1776.35  5344.6 1776.90  5385.0 1776.42  5409.6 1777.05
#Mann=3,-1,0
  4262.7    0.05       0  4987.7    0.05       0  4995.3    0.05       0
Bank Sta=4987.7,4995.3
Exp/Cntr=0.3,0.1

Type RM Length L Ch R = 1,5563,150,150,150
BEGIN DESCRIPTION:
Elm 02 17 5562.87
END DESCRIPTION:
XS GIS Cut Line= 3
      1613048.25      6834909.86      1613505.23      6834912.46
      1613856.82      6834908.56
#Sta/Elev= 30
  4542.8 1772.47  4569.6 1771.61  4609.6 1771.44  4639.6 1769.62  4679.6 1768.14
  4699.6 1767.83  4719.6 1767.94  4739.6 1768.67  4789.6 1769.66  4809.6 1768.91
  4829.6 1768.78  4879.6 1769.41  4919.6 1768.72  4939.6 1769.43  4949.6 1768.94
  4969.6 1766.29  4985.8 1766.04  4986.3 1765.54  4992.9 1765.54  4993.4 1766.04
  5009.6 1766.06  5029.6 1766.55  5049.6 1768.46  5059.6 1768.40  5159.6 1771.45
  5169.6 1771.97  5189.6 1774.21  5219.6 1774.29  5289.6 1775.79  5351.4 1776.73
#Mann=3,-1,0
  4542.8    0.05       0  4985.8    0.05       0  4993.4    0.05       0
Bank Sta=4985.8,4993.4
Exp/Cntr=0.3,0.1

Type RM Length L Ch R = 1,5413,367,367,367
BEGIN DESCRIPTION:
Elm 02 17 5413.46
END DESCRIPTION:
XS GIS Cut Line= 3
      1613057.28      6835040.07      1613415.39      6835027.05
      1613881.44      6835027.05
#Sta/Elev= 30
  4641.8 1768.11  4699.6 1767.15  4739.6 1767.38  4749.6 1767.74  4819.6 1768.00
  4835.5 1766.57  4840.5 1767.62  4849.7 1766.69  4859.7 1766.53  4899.7 1766.94
  4929.7 1766.00  4955.9 1765.90  4956.4 1765.40  4963.0 1765.40  4963.5 1765.90
  5009.8 1768.57  5039.8 1769.17  5049.8 1768.97  5069.8 1769.25  5119.8 1770.25
  5139.8 1770.86  5159.8 1772.35  5169.8 1772.34  5179.8 1772.77  5219.8 1772.88
  5229.8 1773.35  5289.8 1774.23  5309.8 1775.14  5359.8 1776.30  5466.2 1777.74
#Mann=3,-1,0
  4641.8    0.05       0  4955.9    0.05       0  4963.5    0.05       0
Bank Sta=4955.9,4963.5
Exp/Cntr=0.3,0.1

Type RM Length L Ch R = 1,5046,267,267,267
BEGIN DESCRIPTION:
Elm 02 17 5143.66
END DESCRIPTION:
XS GIS Cut Line= 3
      1612994.82      6835015.34      1613106.58      6835191.83
      1613346.38      6835601.27
#Sta/Elev= 30
  4791.1 1769.68  4800.5 1769.79  4806.4 1769.52  4815.7 1768.56  4836.9 1767.74
  4842.8 1767.93  4858.1 1767.80  4865.3 1767.50  4909.8 1767.22  4931.0 1766.47
  4936.9 1766.61  4982.7 1766.26  4994.8 1763.37  5014.9 1763.00  5015.4 1762.50
  5022.1 1762.50  5022.6 1763.00  5025.5 1763.00  5031.3 1763.95  5041.2 1764.99
  5047.0 1765.09  5053.5 1766.87  5068.5 1768.59  5185.8 1768.64  5215.8 1769.45
  5238.7 1769.23  5303.1 1769.36  5308.9 1769.62  5398.9 1770.23  5474.5 1771.15
#Mann=3,-1,0
  4791.1    0.05       0  5014.9    0.03       0  5022.6    0.05       0
Bank Sta=5014.9,5022.6
Exp/Cntr=0.3,0.1

Type RM Length L Ch R = 1,4779,475,475,475
BEGIN DESCRIPTION:
Elm 02 17 4778.92
END DESCRIPTION:
XS GIS Cut Line= 3
      1612876.54      6835024.97      1612870.03      6835289.70
      1612941.65      6835751.97
#Sta/Elev= 30
  4736.9 1769.97  4769.9 1769.10  4779.9 1769.28  4799.9 1768.17  4810.0 1768.28
  4820.0 1767.50  4850.0 1766.38  4920.0 1765.63  4990.0 1763.01  4998.4 1763.26
  5010.1 1763.09  5030.3 1765.10  5040.5 1765.28  5060.7 1764.85  5066.3 1764.24
  5080.9 1764.00  5107.5 1762.98  5108.0 1762.48  5114.7 1762.48  5115.2 1762.98
  5121.4 1763.05  5141.7 1765.74  5151.8 1766.41  5182.1 1767.08  5222.6 1766.81
  5242.9 1767.42  5265.5 1767.14  5391.5 1768.71  5396.6 1768.55  5469.5 1769.36
#Mann=3,-1,0
  4736.9    0.05       0  5107.5    0.05       0  5115.2    0.05       0
Bank Sta=5107.5,5115.2
Exp/Cntr=0.3,0.1

Type RM Length L Ch R = 1,4304,467,467,467
BEGIN DESCRIPTION:
Elm 02 17 4304.13
END DESCRIPTION:
XS GIS Cut Line= 3
      1612600.92      6835142.16      1612444.68      6835443.78
      1612266.75      6835810.51
#Sta/Elev= 30
  4666.8 1765.51  4751.2 1763.38  4778.9 1763.42  4831.0 1762.75  4876.1 1763.33
  4884.0 1762.97  4898.6 1763.16  4906.1 1762.56  4956.0 1761.45  4966.2 1760.87
  4972.5 1759.34  4978.1 1759.63  4988.7 1758.12  4996.4 1757.78  4996.9 1757.28
  5003.7 1757.28  5004.2 1757.78  5006.0 1759.06  5011.6 1759.06  5017.0 1760.62
  5055.6 1762.35  5062.1 1763.01  5084.7 1763.79  5112.8 1763.99  5135.4 1765.09
  5211.2 1765.26  5225.7 1764.93  5287.8 1765.38  5338.5 1764.95  5414.1 1764.85
#Mann=3,-1,0
  4666.8    0.05       0  4996.4    0.05       0  5004.2    0.05       0
Bank Sta=4996.4,5004.2
Exp/Cntr=0.3,0.1

Type RM Length L Ch R = 1,3837,214,214,214
BEGIN DESCRIPTION:
Elm 02 17 3836.75
END DESCRIPTION:
XS GIS Cut Line= 3
      1612655.22      6835064.01      1612195.12      6835083.54
      1611741.55      6835087.88
#Sta/Elev= 30
  4541.3 1767.45  4631.6 1766.21  4651.6 1765.27  4661.6 1765.42  4691.7 1764.75
  4701.7 1764.14  4721.7 1763.91  4741.7 1764.31  4755.0 1763.74  4821.8 1763.12
  4851.8 1762.22  4871.8 1762.49  4881.8 1761.77  4891.8 1762.20  4901.8 1761.81
  4911.9 1762.02  4941.9 1760.46  4951.9 1759.50  4961.9 1757.96  4988.0 1757.10
  5008.0 1756.83  5008.5 1756.33  5015.3 1756.33  5015.8 1756.83  5051.9 1759.47
  5061.9 1761.47  5281.9 1761.85  5311.9 1761.25  5362.0 1761.11  5455.4 1760.04
#Mann=3,-1,0
  4541.3    0.05       0  5008.0    0.05       0  5015.8    0.05       0
Bank Sta=5008,5015.8
Exp/Cntr=0.3,0.1

Type RM Length L Ch R = 1,3623,543,543,543
BEGIN DESCRIPTION:
Elm 02 17 3623.38
END DESCRIPTION:
XS GIS Cut Line= 3
      1612603.14      6834853.50      1612112.65      6834899.08
      1611752.39      6834912.10
#Sta/Elev= 30
  4509.0 1771.76  4517.2 1771.35  4567.4 1770.17  4607.1 1768.93  4647.7 1767.20
  4697.9 1765.65  4728.1 1764.39  4798.4 1762.98  4830.7 1762.94  4838.6 1762.70
  4848.6 1761.82  4898.8 1760.53  4928.9 1760.75  4934.9 1759.57  4939.9 1758.91
  4949.0 1757.93  4959.1 1757.33  4965.2 1756.25  4965.7 1755.75  4972.6 1755.75
  4973.1 1756.25  4979.2 1756.47  5019.3 1756.47  5039.3 1756.74  5049.3 1757.27
  5059.3 1758.51  5069.3 1758.96  5099.3 1758.64  5179.4 1758.89  5362.1 1757.53
#Mann=3,-1,0
  4509.0    0.05       0  4965.2    0.05       0  4973.1    0.05       0
Bank Sta=4965.2,4973.1
Exp/Cntr=0.3,0.1

Type RM Length L Ch R = 1,3080,176,176,176
BEGIN DESCRIPTION:
Elm 02 17 3079.98
END DESCRIPTION:
XS GIS Cut Line= 3
      1611660.65      6834210.82      1611667.17      6834744.68
      1611669.33      6835393.28
#Sta/Elev= 30
  4469.6 1765.36  4646.8 1761.30  4706.8 1760.24  4766.8 1759.80  4866.8 1758.42
  4896.8 1758.70  4956.8 1758.23  4966.8 1757.01  4972.9 1755.06  4973.4 1754.56
  4980.3 1754.56  4980.8 1755.06  4996.8 1757.58  5002.7 1755.99  5016.8 1755.57
  5026.8 1755.96  5066.8 1756.41  5116.8 1756.48  5176.8 1757.15  5236.8 1757.48
  5246.8 1758.36  5256.8 1758.45  5266.8 1758.25  5276.8 1757.54  5296.8 1758.43
  5336.8 1758.56  5446.8 1760.47  5506.8 1761.05  5546.8 1761.26  5652.1 1760.92
#Mann=3,-1,0
  4469.6    0.05       0  4972.9    0.05       0  4980.8    0.05       0
Bank Sta=4972.9,4980.8
Exp/Cntr=0.3,0.1

Type RM Length L Ch R = 1,2904,347,347,347
BEGIN DESCRIPTION:
Elm 02 17 2903.95
END DESCRIPTION:
XS GIS Cut Line= 3
      1611474.02      6834193.43      1611506.58      6834796.77
      1611500.06      6835419.62
#Sta/Elev= 30
  4400.8 1764.92  4475.5 1764.13  4511.1 1762.92  4575.6 1761.60  4595.7 1761.62
  4605.7 1760.58  4635.7 1760.15  4665.8 1758.42  4735.9 1757.23  4876.1 1756.80
  4916.1 1757.13  4956.2 1756.54  4976.2 1757.24  4986.2 1756.66  5003.1 1753.52
  5012.3 1753.06  5012.8 1752.56  5019.7 1752.56  5020.2 1753.06  5026.2 1754.10
  5036.2 1754.47  5066.3 1753.69  5086.3 1755.09  5096.3 1756.33  5136.3 1755.67
  5186.3 1756.33  5306.3 1755.69  5376.3 1756.52  5506.3 1759.47  5627.9 1759.24
#Mann=3,-1,0
  4400.8    0.05       0  5012.3    0.05       0  5020.2    0.05       0
Bank Sta=5012.3,5020.2
Exp/Cntr=0.3,0.1

Type RM Length L Ch R = 1,2557,420,420,420
BEGIN DESCRIPTION:
Elm 02 17 2557.18
END DESCRIPTION:
XS GIS Cut Line= 3
      1611218.81      6834217.90      1611231.84      6834991.35
      1611439.35      6835494.58
#Sta/Elev= 30
  4229.8 1761.90  4249.9 1762.03  4259.9 1761.38  4279.9 1761.61  4297.6 1760.48
  4359.9 1760.05  4399.9 1758.67  4449.9 1758.22  4509.9 1756.63  4549.9 1756.88
  4620.0 1755.77  4670.0 1756.16  4880.0 1754.72  4920.0 1754.78  4970.0 1755.75
  4980.0 1754.91  4999.2 1751.20  5003.4 1751.20  5006.6 1750.38  5007.1 1749.88
  5014.1 1749.88  5014.6 1750.38  5020.4 1750.44  5043.0 1752.66  5055.1 1755.24
  5226.9 1753.48  5340.0 1754.91  5454.0 1757.79  5499.8 1758.45  5547.7 1758.52
#Mann=3,-1,0
  4229.8    0.05       0  5006.6    0.05       0  5014.6    0.05       0
Bank Sta=5006.6,5014.6
Exp/Cntr=0.3,0.1

Type RM Length L Ch R = 1,2137,470,470,470
BEGIN DESCRIPTION:
Elm 02 17 2137.27
END DESCRIPTION:
XS GIS Cut Line= 3
      1610966.21      6834361.12      1610877.67      6835191.88
      1611725.84      6836073.87
#Sta/Elev= 30
  4168.0 1758.59  4205.1 1758.61  4255.4 1757.09  4446.4 1754.87  4557.1 1755.12
  4838.7 1752.58  4899.0 1753.14  4929.2 1752.08  4959.3 1752.13  4973.9 1749.05
  4974.4 1748.55  4982.0 1749.05  5020.1 1750.01  5027.0 1750.76  5034.2 1752.58
  5048.4 1751.06  5175.7 1752.61  5331.1 1752.09  5423.2 1753.12  5451.5 1753.84
  5465.7 1755.04  5529.2 1756.37  5691.8 1756.76  5762.5 1755.55  5805.0 1756.67
  5889.9 1756.21  5982.0 1757.69  5988.9 1759.54  6031.4 1760.18  6227.1 1760.71
#Mann=3,-1,0
  4168.0    0.05       0  4973.9    0.05       0  4982.0    0.05       0
Bank Sta=4973.9,4982
Exp/Cntr=0.3,0.1

Type RM Length L Ch R = 1,1667,0,0,0
BEGIN DESCRIPTION:
Elm 02 17 1666.77
END DESCRIPTION:
XS GIS Cut Line= 4
      1610806.83      6834358.28      1610470.01      6835399.99
      1610650.57      6836007.63      1611775.56      6836212.49
#Sta/Elev= 30
  3917.2 1759.59  4022.0 1758.26  4043.0 1758.64  4101.4 1757.04  4158.6 1756.61
  4179.6 1756.99  4242.7 1755.39  4752.2 1752.41  4799.7 1751.73  4816.3 1750.75
  4862.8 1749.89  4957.4 1750.33  4981.6 1751.07  5004.2 1744.73  5004.7 1744.23
  5011.9 1744.23  5012.4 1744.73  5041.2 1750.90  5062.1 1749.45  5085.2 1749.14
  5385.5 1748.00  5448.1 1748.78  5499.2 1748.39  5787.6 1749.23  6168.8 1752.44
  6511.2 1758.82  6544.9 1759.01  6605.9 1761.17  6681.4 1760.73  6789.4 1761.55
#Mann=3,-1,0
  3917.2    0.05       0  5004.2    0.05       0  5012.4    0.05       0
Bank Sta=5004.2,5012.4
Exp/Cntr=0.3,0.1

Chan Stop Cuts=-1
