--- Elm 02 31.prj (project) ---

Proj Title=Elm 02 31 Base Level Engineering
Current Plan=p01
Default Exp/Contr=0.3,0.1
English Units
Geom File=g01
Flow File=f01
Plan File=p01
BEGIN DESCRIPTION:
Elm 02 31
END DESCRIPTION:

--- Elm 02 31.p01 (plan) ---

Plan Title=Multiple Run
Short Identifier=Multiple
Geom File=g01
Flow File=f01
Subcritical Flow
K Sum by GR= 0
Std Step Tol= 0.01
Critical Tol= 0.01
Num of Std Step Trials= 20
Max Error Tol= 0.3
Flow Tol Ratio= 0.001
Split Flow NTrial= 30
Split Flow Tol= 0.02
Split Flow Ratio= 0.02
Log Output Level= 0
Friction Slope Method= 1
Unsteady Friction Slope Method= 2
Unsteady Bridges Friction Slope Method= 1
Parabolic Critical Depth
Global Vel Dist=  1 , 1 , 1
Global Log Level= 0
CheckData=True
Encroach Param= -1, 0, 0, 0
BEGIN DESCRIPTION:
Multiple Run
END DESCRIPTION:

--- Elm 02 31.f01 (steady flow) ---

Flow Title=Multiple
Number of Profiles=7
Profile Names=10-year,25-year,50-year,1pct_min,100-year,1pct_plu,500-year
River Rch & RM= Elm 02 31,Reach-1,11181
     197     269     328     248     398     547     591
River Rch & RM= Elm 02 31,Reach-1,4223
     286     399     493     377     605     832     923
River Rch & RM= Elm 02 31,Reach-1,16
    2270    3400    4400    3500    5610    7720    9270
Boundary for River Rch & Prof#=Elm 02 31,Reach-1,1
Up Type=0
Dn Type=3
Dn Slope=0.001
Boundary for River Rch & Prof#=Elm 02 31,Reach-1,2
Up Type=0
Dn Type=3
Dn Slope=0.001
Boundary for River Rch & Prof#=Elm 02 31,Reach-1,3
Up Type=0
Dn Type=3
Dn Slope=0.001
Boundary for River Rch & Prof#=Elm 02 31,Reach-1,4
Up Type=0
Dn Type=3
Dn Slope=0.001
Boundary for River Rch & Prof#=Elm 02 31,Reach-1,5
Up Type=0
Dn Type=3
Dn Slope=0.001
Boundary for River Rch & Prof#=Elm 02 31,Reach-1,6
Up Type=0
Dn Type=3
Dn Slope=0.001
Boundary for River Rch & Prof#=Elm 02 31,Reach-1,7
Up Type=0
Dn Type=3
Dn Slope=0.001

--- Elm 02 31.g01 (geometry) ---

Geom Title=Existing Conditions

River Reach=Elm 02 31,Reach-1
Reach XY= 30
      1606605.00      6858088.00      1606378.57      6858515.14
      1605995.21      6858648.52      1605858.13      6858789.63
      1605835.25      6859008.42      1605594.90      6859098.39
      1605457.46      6859282.54      1605144.84      6859348.36
      1605053.75      6859584.49      1604720.22      6859637.48
      1604270.22      6859488.23      1604103.54      6859634.46
      1603852.53      6859643.46      1603743.17      6859786.38
      1603529.91      6859788.21      1603203.48      6859441.74
      1602848.57      6859496.02      1602851.55      6859836.75
      1602611.19      6860080.15      1602106.55      6860141.75
      1601899.15      6860336.46      1601628.13      6860314.16
      1601160.30      6860785.33      1601253.39      6861081.97
      1601011.19      6861330.19      1600710.86      6861335.94
      1600504.91      6861195.28      1600303.54      6861384.46
      1599941.33      6861401.23      1599105.00      6862738.00

Type RM Length L Ch R = 1,11181,160,160,160
BEGIN DESCRIPTION:
Elm 02 31 10861.478
END DESCRIPTION:
XS GIS Cut Line= 3
      1606423.49      6857909.47      1606586.60      6858107.17
      1606819.34      6858336.58
#Sta/Elev= 30
  4743.7 1734.15  4771.9 1734.31  4779.8 1733.84  4786.3 1734.18  4793.6 1733.85
  4858.0 1733.61  4885.3 1733.17  4893.1 1732.66  4899.6 1732.91  4928.3 1732.39
  4977.8 1730.89  5011.6 1729.10  5011.8 1728.60  5015.3 1728.60  5015.6 1729.10
  5027.7 1729.37  5034.8 1730.33  5041.8 1730.25  5049.0 1730.83  5056.0 1730.52
  5063.1 1730.84  5084.3 1730.69  5105.5 1731.87  5112.6 1731.55  5119.7 1732.10
  5162.1 1733.22  5261.1 1734.57  5282.3 1734.49  5303.5 1735.04  5326.8 1734.92
#Mann=3,-1,0
  4743.7    0.05       0  5011.6    0.05       0  5015.6    0.05       0
Bank Sta=5011.6,5015.6
Exp/Cntr=0.3,0.1

Type RM Length L Ch R = 1,11021,275,275,275
BEGIN DESCRIPTION:
Elm 02 31 11021.09
END DESCRIPTION:
XS GIS Cut Line= 3
      1606315.85      6858043.16      1606508.58      6858241.09
      1606734.91      6858413.86
#Sta/Elev= 30
  4723.8 1731.50  4761.9 1731.79  4846.8 1730.79  4861.0 1731.00  4868.1 1730.42
  4938.9 1729.17  4960.0 1727.60  4988.3 1726.00  5000.1 1725.87  5000.5 1725.59
  5000.8 1725.09  5004.3 1725.09  5004.5 1725.59  5037.9 1725.95  5045.9 1726.27
  5052.4 1726.99  5058.7 1726.66  5066.9 1727.33  5073.2 1727.20  5081.5 1728.07
  5096.0 1728.86  5102.3 1728.79  5116.8 1729.54  5152.2 1730.42  5181.2 1731.70
  5202.1 1731.68  5231.1 1732.68  5251.9 1732.34  5266.5 1732.97  5284.8 1732.69
#Mann=3,-1,0
  4723.8    0.05       0  5000.5    0.03       0  5004.5    0.05       0
Bank Sta=5000.5,5004.5
Exp/Cntr=0.3,0.1

Type RM Length L Ch R = 1,10746,218,218,218
BEGIN DESCRIPTION:
Elm 02 31 10746.2
END DESCRIPTION:
XS GIS Cut Line= 3
      1606188.09      6858162.93      1606410.30      6858485.82
      1606755.25      6858813.44
#Sta/Elev= 30
  4609.9 1728.29  4617.7 1728.61  4676.8 1728.54  4698.2 1728.16  4719.2 1728.54
  4761.7 1727.55  4790.9 1727.46  4820.6 1726.18  4826.7 1726.30  4919.5 1723.24
  4949.1 1722.84  4990.4 1721.60  4990.6 1721.10  4994.1 1721.10  4994.4 1721.60
  5013.8 1721.71  5063.5 1723.22  5070.4 1722.98  5098.7 1724.20  5127.0 1724.86
  5169.5 1725.04  5197.8 1726.13  5204.7 1725.77  5226.1 1726.03  5325.2 1729.07
  5353.1 1729.37  5402.9 1730.82  5409.8 1730.57  5431.2 1731.11  5477.6 1731.38
#Mann=3,-1,0
  4609.9    0.05       0  4990.4    0.03       0  4994.4    0.05       0
Bank Sta=4990.4,4994.4
Exp/Cntr=0.3,0.1

Type RM Length L Ch R = 1,10528,321,321,321
BEGIN DESCRIPTION:
Elm 02 31 10527.92
END DESCRIPTION:
XS GIS Cut Line= 5
      1606135.70      6858102.49      1606153.06      6858486.61
      1606221.19      6858570.50      1606307.14      6858629.84
      1606524.58      6858675.97
#Sta/Elev= 30
  4507.4 1727.31  4573.0 1727.50  4600.3 1727.11  4605.3 1727.37  4623.0 1726.88
  4663.1 1726.81  4703.1 1726.24  4713.1 1725.82  4763.2 1724.96  4773.2 1724.29
  4821.1 1722.64  4826.1 1723.08  4890.1 1720.21  4951.1 1719.82  4965.5 1719.30
  4971.9 1719.44  4979.8 1718.85  4992.2 1718.73  4992.5 1718.23  4996.0 1718.23
  4996.2 1718.73  5007.5 1718.78  5037.3 1719.66  5058.2 1720.74  5088.0 1721.49
  5104.4 1721.55  5132.9 1722.48  5163.1 1722.88  5168.3 1723.35  5326.7 1725.92
#Mann=3,-1,0
  4507.4    0.05       0  4992.2    0.05       0  4996.2    0.05       0
Bank Sta=4992.2,4996.2
Exp/Cntr=0.3,0.1

Type RM Length L Ch R = 1,10207,167,167,167
BEGIN DESCRIPTION:
Elm 02 31 10207.31
END DESCRIPTION:
XS GIS Cut Line= 5
      1605415.18      6858657.74      1605943.85      6858699.41
      1606087.08      6858679.87      1606191.24      6858639.51
      1606540.06      6858709.79
#Sta/Elev= 30
  4469.8 1724.02  4535.8 1723.84  4620.1 1722.48  4659.6 1722.71  4670.2 1722.13
  4700.3 1722.59  4840.8 1720.72  4870.9 1719.25  4917.3 1717.81  4922.3 1718.25
  4941.1 1718.37  4951.1 1717.63  4961.1 1716.12  4981.2 1715.24  4998.2 1713.80
  5151.2 1713.52  5151.4 1713.02  5154.9 1713.02  5155.2 1713.52  5166.5 1713.79
  5191.0 1716.31  5196.4 1715.99  5215.6 1718.35  5245.5 1719.47  5250.9 1719.14
  5280.6 1719.74  5433.6 1723.89  5472.9 1724.21  5478.0 1724.64  5612.2 1726.96
#Mann=3,-1,0
  4469.8    0.05       0  5151.2    0.05       0  5155.2    0.05       0
Bank Sta=5151.2,5155.2
Exp/Cntr=0.3,0.1

Type RM Length L Ch R = 1,10040,328,328,328
BEGIN DESCRIPTION:
Elm 02 31 10039.61
END DESCRIPTION:
XS GIS Cut Line= 5
      1605380.02      6858821.80      1605856.61      6858832.22
      1606049.32      6858838.73      1606176.92      6858800.97
      1606556.29      6858823.05
#Sta/Elev= 30
  4522.9 1721.10  4717.9 1720.10  4747.9 1720.49  4838.0 1719.90  5036.0 1715.59
  5036.3 1715.09  5039.8 1715.09  5040.0 1715.59  5048.0 1715.90  5058.0 1716.92
  5078.0 1722.63  5088.0 1724.04  5108.1 1725.41  5219.2 1725.28  5279.8 1726.65
  5285.0 1725.95  5292.2 1726.64  5313.1 1727.60  5333.6 1727.37  5359.5 1728.37
  5364.5 1728.25  5373.7 1726.34  5383.7 1723.40  5403.7 1722.91  5463.8 1724.43
  5473.8 1724.30  5574.0 1726.26  5624.1 1726.72  5674.2 1727.86  5705.5 1728.02
#Mann=3,-1,0
  4522.9    0.05       0  5036.0    0.03       0  5040.0    0.05       0
Bank Sta=5036,5040
Exp/Cntr=0.3,0.1

Type RM Length L Ch R = 1,9712,274,274,274
BEGIN DESCRIPTION:
Elm 02 31 9711.68
END DESCRIPTION:
XS GIS Cut Line= 3
      1605571.45      6858901.88      1605739.42      6859054.22
      1606034.96      6859249.51
#Sta/Elev= 30
  4772.6 1719.39  4793.4 1718.55  4800.8 1718.83  4815.0 1718.00  4821.8 1718.05
  4829.2 1717.37  4843.4 1717.07  4878.6 1715.47  4949.5 1714.06  4956.3 1713.83
  4961.7 1713.25  4962.0 1712.75  4965.5 1712.75  4965.7 1713.25  4977.9 1713.28
  4998.5 1714.08  5006.1 1713.80  5034.7 1713.90  5070.8 1714.71  5113.9 1715.22
  5122.0 1715.79  5179.2 1716.68  5194.3 1717.40  5251.4 1717.70  5266.5 1718.22
  5287.4 1718.14  5302.6 1718.79  5323.7 1718.38  5329.7 1718.73  5353.6 1718.82
#Mann=3,-1,0
  4772.6    0.05       0  4961.7    0.03       0  4965.7    0.05       0
Bank Sta=4961.7,4965.7
Exp/Cntr=0.3,0.1

Type RM Length L Ch R = 1,9438,252,252,252
BEGIN DESCRIPTION:
Elm 02 31 9438.29
END DESCRIPTION:
XS GIS Cut Line= 3
      1605373.53      6858980.00      1605545.41      6859198.75
      1605779.24      6859563.79
#Sta/Elev= 30
  4723.5 1717.90  4815.6 1716.26  4830.1 1715.58  4844.5 1715.63  4908.7 1713.94
  4915.0 1714.16  4937.2 1713.24  4958.4 1712.87  4972.8 1711.65  4991.7 1711.01
  4991.9 1710.51  4995.4 1710.51  4995.7 1711.01  4998.0 1711.31  5008.5 1711.43
  5014.4 1711.84  5029.6 1712.08  5044.8 1711.72  5060.0 1712.50  5081.2 1712.26
  5095.8 1712.45  5159.8 1714.46  5226.4 1715.30  5247.7 1715.94  5262.1 1715.97
  5268.9 1716.39  5274.8 1716.15  5333.3 1716.96  5392.7 1717.17  5435.2 1717.65
#Mann=3,-1,0
  4723.5    0.05       0  4991.7    0.03       0  4995.7    0.05       0
Bank Sta=4991.7,4995.7
Exp/Cntr=0.3,0.1

Type RM Length L Ch R = 1,9186,214,214,214
BEGIN DESCRIPTION:
Elm 02 31 9186.07
END DESCRIPTION:
XS GIS Cut Line= 3
      1605245.23      6859110.19      1605328.56      6859291.16
      1605430.05      6859568.32
#Sta/Elev= 30
  4803.0 1715.95  4815.8 1715.90  4822.6 1715.44  4844.6 1714.81  4861.7 1713.90
  4867.2 1714.07  4913.1 1712.84  4921.7 1711.98  4930.6 1711.58  4936.1 1711.65
  4953.5 1710.81  4959.0 1710.71  4965.7 1711.09  4982.0 1710.85  4997.7 1709.86
  5002.2 1709.86  5003.3 1709.29  5003.6 1708.79  5007.1 1708.79  5007.3 1709.29
  5020.2 1709.81  5030.5 1710.63  5035.8 1710.48  5105.4 1711.73  5122.0 1711.82
  5213.6 1713.84  5222.5 1713.75  5254.5 1714.20  5286.4 1714.39  5297.4 1714.66
#Mann=3,-1,0
  4803.0    0.05       0  5003.3    0.03       0  5007.3    0.05       0
Bank Sta=5003.3,5007.3
Exp/Cntr=0.3,0.1

Type RM Length L Ch R = 1,8972,227,227,227
BEGIN DESCRIPTION:
Elm 02 31 8972.16
END DESCRIPTION:
XS GIS Cut Line= 3
      1605032.22      6859239.22      1605136.35      6859358.98
      1605311.09      6859586.78
#Sta/Elev= 30
  4843.0 1713.81  4879.9 1713.09  4894.2 1713.19  4907.6 1712.81  4921.7 1712.90
  4929.3 1712.44  4943.5 1711.95  4950.2 1711.96  4986.3 1709.73  4992.9 1709.01
  4995.7 1708.11  4996.0 1707.61  4999.5 1707.61  4999.7 1708.11  5004.2 1708.11
  5007.2 1708.60  5021.7 1709.14  5028.0 1709.63  5050.8 1709.36  5057.1 1709.54
  5071.6 1709.44  5077.9 1709.66  5136.0 1710.01  5142.3 1710.38  5156.8 1710.22
  5206.6 1711.71  5221.2 1711.85  5271.0 1713.07  5285.5 1713.01  5288.8 1713.27
#Mann=3,-1,0
  4843.0    0.05       0  4995.7    0.03       0  4999.7    0.05       0
Bank Sta=4995.7,4999.7
Exp/Cntr=0.3,0.1

Type RM Length L Ch R = 1,8745,249,249,249
BEGIN DESCRIPTION:
Elm 02 31 8744.5
END DESCRIPTION:
XS GIS Cut Line= 3
      1604902.53      6859354.60      1605077.91      6859566.44
      1605198.14      6859694.41
#Sta/Elev= 30
  4725.2 1711.58  4757.3 1711.14  4765.2 1710.81  4771.7 1711.10  4779.5 1710.91
  4786.0 1710.98  4829.0 1710.07  4835.5 1710.12  4872.0 1709.42  4878.5 1709.44
  4892.8 1708.85  4899.3 1709.00  4907.1 1708.73  4921.5 1708.60  4950.1 1708.55
  4971.0 1708.74  4991.8 1708.21  4998.0 1706.79  5004.2 1706.62  5004.5 1706.12
  5008.0 1706.12  5008.2 1706.62  5013.5 1707.22  5020.4 1708.76  5034.6 1709.82
  5041.9 1709.62  5056.0 1710.16  5077.1 1710.53  5098.4 1711.31  5175.8 1712.60
#Mann=3,-1,0
  4725.2    0.05       0  5004.2    0.03       0  5008.2    0.05       0
Bank Sta=5004.2,5008.2
Exp/Cntr=0.3,0.1

Type RM Length L Ch R = 1,8496,222,222,222
BEGIN DESCRIPTION:
Elm 02 31 8496.14
END DESCRIPTION:
XS GIS Cut Line= 3
      1604781.47      6859396.09      1604851.99      6859639.14
      1605114.55      6859893.02
#Sta/Elev= 30
  4749.2 1710.47  4824.1 1709.48  4850.8 1708.83  4889.6 1708.27  4923.2 1707.33
  4928.4 1707.56  4961.9 1706.85  4969.8 1706.05  4980.3 1705.57  4990.3 1705.77
  4993.5 1705.50  4993.7 1705.00  4997.2 1705.00  4997.5 1705.50  4999.1 1706.29
  5005.1 1706.29  5010.6 1706.77  5032.0 1707.29  5067.2 1707.56  5145.1 1709.33
  5194.5 1710.23  5201.5 1710.19  5222.8 1710.71  5293.6 1711.04  5300.5 1711.27
  5321.9 1711.28  5328.8 1711.09  5350.2 1711.44  5357.1 1711.23  5367.5 1711.48
#Mann=3,-1,0
  4749.2    0.05       0  4993.5    0.03       0  4997.5    0.05       0
Bank Sta=4993.5,4997.5
Exp/Cntr=0.3,0.1

Type RM Length L Ch R = 1,8274,234,234,234
BEGIN DESCRIPTION:
Elm 02 31 8274.24
END DESCRIPTION:
XS GIS Cut Line= 3
      1604683.82      6859338.53      1604644.75      6859591.40
      1604631.80      6859894.65
#Sta/Elev= 30
  4746.1 1710.53  4796.2 1710.10  4846.8 1709.24  4856.9 1708.86  4867.0 1708.92
  4887.2 1708.45  4897.2 1708.40  4902.2 1708.00  4947.9 1707.23  4965.3 1706.26
  5002.0 1705.87  5008.6 1705.35  5016.6 1704.97  5016.8 1704.47  5020.3 1704.47
  5020.6 1704.97  5028.6 1705.38  5038.6 1706.14  5113.4 1707.29  5138.7 1707.84
  5148.7 1708.24  5178.7 1708.52  5188.7 1708.79  5208.8 1708.64  5218.8 1708.94
  5248.8 1709.33  5258.8 1709.24  5278.8 1709.50  5288.8 1709.43  5305.5 1709.80
#Mann=3,-1,0
  4746.1    0.05       0  5016.6    0.03       0  5020.6    0.05       0
Bank Sta=5016.6,5020.6
Exp/Cntr=0.3,0.1

Type RM Length L Ch R = 1,8040,388,388,388
BEGIN DESCRIPTION:
Elm 02 31 8039.62
END DESCRIPTION:
XS GIS Cut Line= 3
      1604589.40      6859271.32      1604410.37      6859584.89
      1604466.62      6859903.99
#Sta/Elev= 30
  4640.8 1711.04  4657.0 1710.97  4678.6 1710.34  4684.4 1710.46  4706.1 1710.11
  4729.1 1709.43  4752.1 1709.48  4780.8 1709.00  4786.7 1709.12  4824.0 1708.10
  4839.9 1707.24  4861.5 1706.87  4890.3 1705.90  4936.4 1705.31  4993.9 1705.03
  5000.8 1704.47  5006.0 1704.47  5013.2 1704.06  5013.4 1703.56  5016.9 1703.56
  5017.2 1704.06  5025.3 1704.16  5054.0 1705.95  5066.0 1705.91  5126.9 1707.45
  5248.7 1708.62  5279.2 1708.69  5291.1 1708.97  5319.8 1709.04  5325.9 1709.25
#Mann=3,-1,0
  4640.8    0.05       0  5013.2    0.03       0  5017.2    0.05       0
Bank Sta=5013.2,5017.2
Exp/Cntr=0.3,0.1

Type RM Length L Ch R = 1,7652,90,90,90
BEGIN DESCRIPTION:
Elm 02 31 7651.55
END DESCRIPTION:
XS GIS Cut Line= 5
      1604239.22      6859270.43      1604115.52      6859499.60
      1604107.71      6859572.52      1604128.54      6859612.88
      1604379.84      6859796.47
#Sta/Elev= 30
  4619.3 1708.91  4811.3 1705.88  4827.5 1706.76  4833.2 1706.16  4843.7 1707.31
  4849.4 1706.77  4855.2 1708.44  4865.6 1709.24  4871.3 1708.42  4888.2 1709.51
  4932.5 1707.97  4953.1 1708.45  4955.8 1707.85  4961.5 1709.50  4978.0 1708.73
  4983.6 1709.59  4998.5 1708.43  5006.5 1709.01  5028.8 1708.44  5035.0 1707.58
  5043.5 1708.06  5049.7 1706.28  5064.4 1707.21  5070.5 1705.20  5079.0 1705.59
  5083.2 1704.54  5083.5 1704.04  5087.2 1704.54  5221.1 1707.03  5309.7 1707.80
#Mann=3,-1,0
  4619.3    0.05       0  5083.2    0.03       0  5087.2    0.05       0
Bank Sta=5083.2,5087.2
Exp/Cntr=0.3,0.1

Type RM Length L Ch R = 1,7562,264,264,264
BEGIN DESCRIPTION:
Elm 02 31 7562.49
END DESCRIPTION:
XS GIS Cut Line= 3
      1604050.37      6859299.14      1604048.20      6859642.06
      1604152.38      6859828.72
#Sta/Elev= 30
  4660.8 1707.65  4689.7 1706.93  4709.7 1706.86  4716.7 1706.41  4721.7 1706.51
  4739.7 1706.06  4769.7 1705.66  4779.7 1705.73  4789.7 1705.25  4819.7 1705.10
  4839.7 1704.77  4859.7 1704.37  4869.7 1703.94  4889.7 1703.45  4909.7 1703.11
  4939.7 1703.14  4959.7 1702.88  4967.7 1702.48  4967.9 1701.98  4971.4 1701.98
  4971.7 1702.48  4989.7 1702.81  5006.1 1702.62  5027.8 1703.35  5114.7 1705.16
  5124.9 1705.08  5130.7 1705.44  5136.5 1705.04  5152.4 1705.43  5217.5 1706.24
#Mann=3,-1,0
  4660.8    0.05       0  4967.7    0.03       0  4971.7    0.05       0
Bank Sta=4967.7,4971.7
Exp/Cntr=0.3,0.1

Type RM Length L Ch R = 1,7298,251,251,251
BEGIN DESCRIPTION:
Elm 02 31 7297.8
END DESCRIPTION:
XS GIS Cut Line= 3
      1603792.12      6859227.58      1603802.97      6859694.14
      1603972.25      6860063.07
#Sta/Elev= 30
  4537.1 1706.11  4577.5 1705.44  4587.5 1705.60  4607.5 1705.53  4637.5 1705.02
  4677.6 1705.22  4707.6 1704.59  4717.6 1704.61  4777.6 1703.80  4827.6 1703.49
  4847.6 1703.13  4879.3 1703.01  4957.6 1702.13  4967.6 1701.77  4977.6 1700.80
  4985.6 1700.60  4985.9 1700.10  4989.4 1700.10  4989.6 1700.60  4997.6 1701.53
  5068.6 1701.48  5212.0 1704.77  5258.0 1705.32  5272.1 1705.68  5281.0 1705.66
  5316.1 1706.66  5361.0 1707.19  5378.5 1707.63  5393.1 1707.66  5409.7 1708.18
#Mann=3,-1,0
  4537.1    0.05       0  4985.6    0.05       0  4989.6    0.05       0
Bank Sta=4985.6,4989.6
Exp/Cntr=0.3,0.1

Type RM Length L Ch R = 1,7047,191,191,191
BEGIN DESCRIPTION:
Elm 02 31 7047.42
END DESCRIPTION:
XS GIS Cut Line= 3
      1603681.44      6859448.92      1603609.83      6859791.80
      1603583.79      6860089.08
#Sta/Elev= 30
  4653.2 1703.15  4663.9 1703.01  4672.7 1703.33  4693.1 1702.61  4753.7 1702.20
  4774.9 1701.70  4815.7 1701.56  4825.9 1701.25  4853.7 1700.99  4897.4 1701.03
  4908.8 1700.79  4953.7 1700.91  4958.8 1701.08  4979.2 1700.64  5007.7 1699.46
  5008.0 1698.96  5011.5 1698.96  5011.7 1699.46  5039.8 1700.01  5049.9 1700.94
  5069.9 1701.68  5100.1 1702.26  5115.6 1702.90  5130.2 1703.24  5160.3 1703.77
  5220.5 1704.28  5228.1 1704.51  5233.1 1704.40  5240.6 1704.62  5301.9 1705.05
#Mann=3,-1,0
  4653.2    0.05       0  5007.7    0.03       0  5011.7    0.05       0
Bank Sta=5007.7,5011.7
Exp/Cntr=0.3,0.1

Type RM Length L Ch R = 1,6856,230,230,230
BEGIN DESCRIPTION:
Elm 02 31 6855.72
END DESCRIPTION:
XS GIS Cut Line= 5
      1603640.06      6859410.62      1603520.89      6859674.78
      1603431.73      6859740.17      1603345.66      6859828.09
      1603284.33      6859993.49
#Sta/Elev= 30
  4602.5 1703.20  4627.0 1702.60  4678.7 1702.25  4687.4 1701.99  4731.3 1701.79
  4742.2 1701.50  4748.1 1701.58  4851.9 1700.28  4935.3 1699.98  4949.2 1699.45
  4962.4 1699.78  4977.0 1699.75  5002.9 1699.30  5006.1 1698.63  5011.2 1698.39
  5011.5 1697.89  5015.0 1697.89  5015.2 1698.39  5027.4 1699.92  5069.8 1700.93
  5090.9 1701.26  5119.2 1701.05  5167.0 1701.59  5189.8 1701.61  5197.4 1701.93
  5202.7 1701.61  5252.8 1701.96  5264.5 1701.84  5288.5 1702.33  5302.3 1703.35
#Mann=3,-1,0
  4602.5    0.05       0  5011.2    0.03       0  5015.2    0.05       0
Bank Sta=5011.2,5015.2
Exp/Cntr=0.3,0.1

Type RM Length L Ch R = 1,6626,186,186,186
BEGIN DESCRIPTION:
Elm 02 31 6626.42
END DESCRIPTION:
XS GIS Cut Line= 5
      1603534.14      6859318.64      1603401.12      6859487.78
      1603327.57      6859563.30      1603257.18      6859633.69
      1603239.00      6860030.43
#Sta/Elev= 30
  4681.4 1703.04  4780.6 1701.76  4786.9 1701.18  4807.8 1700.68  4815.8 1701.00
  4915.2 1699.44  4964.8 1698.45  4971.8 1697.71  4976.9 1697.66  4977.2 1697.16
  4980.7 1697.16  4980.9 1697.66  4985.9 1698.31  4993.1 1698.37  5007.3 1697.80
  5014.2 1698.28  5021.3 1698.27  5028.3 1698.93  5063.7 1699.06  5070.8 1699.78
  5077.8 1699.16  5106.2 1699.06  5226.0 1699.95  5254.7 1700.47  5326.1 1700.88
  5346.1 1700.69  5356.1 1701.17  5406.2 1701.10  5416.2 1701.45  5498.7 1701.74
#Mann=3,-1,0
  4681.4    0.05       0  4976.9    0.03       0  4980.9    0.05       0
Bank Sta=4976.9,4980.9
Exp/Cntr=0.3,0.1

Type RM Length L Ch R = 1,6440,167,167,167
BEGIN DESCRIPTION:
Elm 02 31 6439.51
END DESCRIPTION:
XS GIS Cut Line= 4
      1603237.26      6859263.13      1603203.87      6859443.94
      1603193.14      6859551.21      1603226.85      6860028.75
#Sta/Elev= 30
  4817.8 1701.19  4863.4 1700.64  4873.6 1701.10  4883.8 1700.59  4893.9 1700.56
  4955.0 1699.00  4969.1 1698.84  4995.6 1697.87  5001.2 1697.31  5013.8 1697.09
  5014.1 1696.59  5017.6 1696.59  5017.8 1697.09  5035.7 1697.91  5040.7 1697.92
  5046.0 1698.22  5056.0 1698.45  5116.3 1698.73  5196.5 1698.55  5216.5 1698.89
  5226.6 1698.83  5256.6 1699.13  5286.7 1699.60  5306.8 1699.55  5316.8 1699.75
  5376.9 1700.15  5397.0 1700.53  5427.1 1700.59  5547.4 1701.53  5588.2 1701.60
#Mann=3,-1,0
  4817.8    0.05       0  5013.8    0.03       0  5017.8    0.05       0
Bank Sta=5013.8,5017.8
Exp/Cntr=0.3,0.1

Type RM Length L Ch R = 1,6273,128,128,128
BEGIN DESCRIPTION:
Elm 02 31 6272.59
END DESCRIPTION:
XS GIS Cut Line= 4
      1603031.34      6859316.99      1603037.85      6859440.69
      1603042.94      6859540.77      1603218.15      6860039.08
#Sta/Elev= 30
  4878.2 1699.86  4919.3 1700.01  4949.3 1699.16  4959.3 1698.29  4996.2 1697.21
  4996.5 1696.71  5000.0 1696.71  5000.2 1697.21  5019.4 1698.07  5029.4 1698.90
  5069.5 1698.75  5098.4 1698.29  5150.4 1698.09  5173.5 1698.29  5181.4 1697.81
  5217.6 1697.88  5248.6 1698.26  5290.1 1698.19  5330.9 1698.59  5336.2 1698.86
  5374.9 1699.31  5392.9 1699.30  5398.2 1699.67  5449.1 1699.94  5460.1 1700.37
  5502.2 1700.31  5587.0 1701.35  5597.6 1701.14  5609.7 1701.52  5630.5 1701.65
#Mann=3,-1,0
  4878.2    0.05       0  4996.2    0.03       0  5000.2    0.05       0
Bank Sta=4996.2,5000.2
Exp/Cntr=0.3,0.1

Type RM Length L Ch R = 1,6145,97,97,97
BEGIN DESCRIPTION:
Elm 02 31 6144.54
END DESCRIPTION:
XS GIS Cut Line= 4
      1602768.73      6859331.07      1602919.58      6859469.99
      1603096.64      6859733.57      1603207.74      6860052.99
#Sta/Elev= 30
  4794.7 1701.54  4839.5 1701.00  4846.3 1699.60  4853.7 1699.22  4860.5 1697.39
  4867.9 1697.28  4874.7 1695.63  4901.0 1694.91  4901.3 1694.41  4904.8 1694.41
  4905.0 1694.91  4924.6 1695.44  4931.4 1696.66  4938.8 1696.90  4945.6 1700.07
  4959.7 1700.12  4966.5 1701.04  4980.7 1699.03  4988.1 1698.55  5089.0 1698.02
  5117.8 1699.22  5140.0 1697.95  5176.0 1698.26  5190.1 1697.69  5212.0 1697.70
  5298.5 1698.07  5420.7 1699.33  5482.9 1700.35  5502.0 1700.17  5655.5 1701.47
#Mann=3,-1,0
  4794.7    0.05       0  4901.0    0.03       0  4905.0    0.05       0
Bank Sta=4901,4905
Exp/Cntr=0.3,0.1

Type RM Length L Ch R = 1,6048,195,195,195
BEGIN DESCRIPTION:
Elm 02 31 6047.76
END DESCRIPTION:
XS GIS Cut Line= 4
      1602679.79      6859389.70      1602836.03      6859510.13
      1603072.33      6859730.10      1603197.34      6860061.71
#Sta/Elev= 30
  4804.0 1701.39  4848.5 1700.57  4877.5 1700.90  4892.0 1699.43  4906.5 1696.49
  4910.8 1696.08  4911.0 1695.58  4914.5 1695.58  4914.8 1696.08  4949.5 1697.52
  4970.8 1697.69  5020.3 1697.68  5034.4 1698.00  5083.8 1698.09  5097.9 1697.80
  5105.3 1698.04  5112.1 1697.71  5147.8 1697.80  5154.6 1697.44  5162.0 1697.88
  5176.1 1697.86  5197.1 1697.24  5225.5 1697.71  5303.1 1697.77  5457.4 1699.98
  5503.5 1699.92  5578.4 1700.76  5627.9 1700.83  5633.2 1701.12  5678.5 1701.49
#Mann=3,-1,0
  4804.0    0.05       0  4910.8    0.05       0  4914.8    0.05       0
Bank Sta=4910.8,4914.8
Exp/Cntr=0.3,0.1

Type RM Length L Ch R = 1,5853,224,224,224
BEGIN DESCRIPTION:
Elm 02 31 5853.07
END DESCRIPTION:
XS GIS Cut Line= 4
      1602641.80      6859627.32      1602853.39      6859677.23
      1603036.59      6859727.51      1603170.63      6860077.34
#Sta/Elev= 30
  4781.9 1699.56  4851.1 1698.82  4867.4 1699.17  4877.7 1698.60  4887.9 1698.84
  4893.4 1698.54  4898.5 1698.97  4908.5 1699.17  4935.7 1697.67  4959.9 1697.03
  4978.1 1697.10  4983.2 1695.33  5009.3 1695.09  5009.6 1694.59  5013.1 1694.59
  5013.3 1695.09  5058.4 1697.05  5125.4 1697.66  5172.1 1697.34  5211.2 1697.95
  5227.0 1698.67  5232.6 1698.26  5251.7 1698.21  5306.4 1698.91  5318.3 1699.57
  5350.4 1700.12  5414.7 1699.87  5481.3 1700.62  5500.4 1700.47  5563.9 1701.45
#Mann=3,-1,0
  4781.9    0.05       0  5009.3    0.03       0  5013.3    0.05       0
Bank Sta=5009.3,5013.3
Exp/Cntr=0.3,0.1

Type RM Length L Ch R = 1,5629,86,86,86
BEGIN DESCRIPTION:
Elm 02 31 5628.71
END DESCRIPTION:
XS GIS Cut Line= 4
      1602701.49      6859699.99      1602778.72      6859855.33
      1602806.50      6859882.24      1603013.07      6860045.41
#Sta/Elev= 30
  4787.9 1698.36  4796.8 1698.49  4804.7 1697.57  4810.3 1698.04  4827.1 1697.37
  4832.7 1697.41  4855.1 1697.02  4886.2 1696.94  4899.9 1696.27  4916.7 1695.09
  4930.9 1694.38  4967.8 1694.50  5065.0 1694.35  5065.3 1693.85  5068.8 1693.85
  5069.0 1694.35  5081.5 1694.38  5087.8 1694.86  5102.3 1696.37  5110.3 1698.53
  5124.8 1700.95  5131.2 1701.51  5138.3 1700.51  5145.6 1698.40  5152.0 1697.26
  5180.8 1697.48  5209.7 1698.08  5216.1 1698.52  5230.5 1698.84  5263.3 1699.16
#Mann=3,-1,0
  4787.9    0.05       0  5065.0    0.05       0  5069.0    0.05       0
Bank Sta=5065,5069
Exp/Cntr=0.3,0.1

Type RM Length L Ch R = 1,5543,74,74,74
BEGIN DESCRIPTION:
Elm 02 31 5542.51
END DESCRIPTION:
XS GIS Cut Line= 5
      1602652.86      6859735.56      1602729.24      6859914.36
      1602759.63      6859957.76      1602825.60      6859985.54
      1602965.32      6860085.34
#Sta/Elev= 30
  4806.6 1698.05  4854.2 1696.36  4894.0 1695.68  4894.2 1695.18  4897.7 1695.18
  4898.0 1695.68  4907.1 1696.68  4925.0 1696.75  4930.4 1698.90  4939.7 1700.08
  4948.6 1700.64  4954.1 1700.24  4972.2 1701.54  4977.7 1700.80  5015.7 1701.07
  5021.8 1700.37  5036.6 1701.55  5042.7 1700.92  5051.1 1701.97  5066.4 1700.73
  5071.8 1701.88  5090.1 1700.77  5095.5 1701.92  5113.9 1700.99  5119.3 1702.02
  5140.9 1702.18  5155.6 1699.30  5161.8 1696.75  5176.5 1696.35  5297.3 1698.87
#Mann=3,-1,0
  4806.6    0.05       0  4894.0    0.05       0  4898.0    0.05       0
Bank Sta=4894,4898
Exp/Cntr=0.3,0.1

Type RM Length L Ch R = 1,5469,310,310,310
BEGIN DESCRIPTION:
Elm 02 31 5469.44
END DESCRIPTION:
XS GIS Cut Line= 5
      1602612.04      6859778.47      1602678.03      6859929.55
      1602703.20      6859979.90      1602762.23      6860036.32
      1602905.46      6860097.08
#Sta/Elev= 30
  4779.6 1697.61  4826.3 1696.93  4844.3 1696.52  4849.7 1695.97  4855.5 1695.72
  4873.1 1695.65  4878.6 1695.17  4888.2 1694.94  4920.0 1695.02  4925.4 1695.24
  4954.2 1694.71  4976.6 1694.62  4993.3 1694.76  4995.2 1694.14  4995.4 1693.64
  4998.9 1693.64  4999.2 1694.14  5021.9 1694.17  5029.1 1694.68  5043.2 1695.05
  5078.5 1694.91  5095.2 1695.21  5100.6 1695.15  5129.7 1695.81  5153.4 1695.86
  5171.6 1696.23  5177.0 1696.68  5194.0 1696.97  5206.1 1697.52  5238.0 1697.86
#Mann=3,-1,0
  4779.6    0.05       0  4995.2    0.05       0  4999.2    0.05       0
Bank Sta=4995.2,4999.2
Exp/Cntr=0.3,0.1

Type RM Length L Ch R = 1,5159,298,298,298
BEGIN DESCRIPTION:
Elm 02 31 5158.5
END DESCRIPTION:
XS GIS Cut Line= 3
      1602323.14      6859857.84      1602455.10      6860135.65
      1602512.38      6860350.90
#Sta/Elev= 30
  4695.9 1696.05  4729.3 1695.49  4786.0 1695.33  4871.4 1693.99  4906.4 1693.97
  4916.8 1693.28  4922.3 1693.45  4928.6 1693.04  4945.1 1692.95  4950.7 1693.41
  4973.3 1693.12  4988.5 1692.43  4988.8 1691.93  4992.3 1691.93  4992.5 1692.43
  5016.2 1692.77  5036.9 1693.57  5047.3 1693.52  5056.9 1693.99  5062.1 1693.87
  5068.0 1694.29  5088.7 1694.80  5097.1 1695.24  5130.1 1695.88  5137.2 1696.47
  5171.5 1698.13  5177.3 1698.91  5182.5 1698.54  5192.2 1699.08  5226.2 1699.19
#Mann=3,-1,0
  4695.9    0.05       0  4988.5    0.05       0  4992.5    0.05       0
Bank Sta=4988.5,4992.5
Exp/Cntr=0.3,0.1

Type RM Length L Ch R = 1,4861,174,174,174
BEGIN DESCRIPTION:
Elm 02 31 4860.62
END DESCRIPTION:
XS GIS Cut Line= 3
      1602001.97      6859887.39      1602156.49      6860137.39
      1602309.25      6860366.54
#Sta/Elev= 30
  4705.9 1695.92  4738.1 1694.93  4774.8 1694.40  4817.3 1694.09  4853.9 1693.41
  4896.5 1693.27  4906.0 1692.84  4918.2 1692.77  4927.2 1692.25  4941.7 1692.08
  4948.5 1691.52  4954.4 1691.57  4963.9 1690.94  4977.0 1690.73  4985.2 1691.11
  5003.0 1691.15  5004.3 1690.73  5004.6 1690.23  5008.1 1690.23  5008.3 1690.73
  5012.5 1691.55  5021.4 1691.84  5057.4 1692.02  5084.7 1692.84  5114.5 1693.11
  5120.7 1693.55  5135.5 1693.39  5144.5 1693.93  5201.6 1694.63  5275.2 1696.27
#Mann=3,-1,0
  4705.9    0.05       0  5004.3    0.05       0  5008.3    0.05       0
Bank Sta=5004.3,5008.3
Exp/Cntr=0.3,0.1

Type RM Length L Ch R = 1,4687,84,84,84
BEGIN DESCRIPTION:
Elm 02 31 4687.41
END DESCRIPTION:
XS GIS Cut Line= 3
      1601590.23      6860064.60      1602001.45      6860197.20
      1602176.13      6860244.71
#Sta/Elev= 30
  4569.7 1694.62  4578.1 1694.63  4616.7 1694.50  4648.3 1693.96  4669.3 1692.72
  4689.9 1692.48  4700.8 1691.83  4764.6 1690.62  4791.3 1690.59  4796.6 1690.31
  4823.4 1690.48  4828.7 1690.22  4855.5 1690.70  4860.7 1690.33  4887.5 1690.48
  4892.8 1690.07  4919.6 1690.30  4924.8 1689.96  4942.5 1690.21  4954.9 1689.95
  4955.1 1689.45  4958.6 1689.45  4958.9 1689.95  5015.8 1689.99  5057.0 1690.74
  5062.2 1691.16  5088.4 1691.19  5129.8 1691.81  5141.8 1692.28  5182.8 1692.56
#Mann=4,-1,0
  4569.7   0.075       0  4578.1    0.05       0  4954.9    0.05       0
  4958.9    0.05       0
Bank Sta=4954.9,4958.9
Exp/Cntr=0.3,0.1

Type RM Length L Ch R = 1,4603,380,380,380
BEGIN DESCRIPTION:
Elm 02 31 4603.3
END DESCRIPTION:
XS GIS Cut Line= 3
      1601590.25      6860168.77      1601955.91      6860263.17
      1602140.23      6860326.05
#Sta/Elev= 30
  4622.9 1693.18  4628.1 1693.18  4636.4 1693.17  4648.5 1692.47  4669.1 1691.84
  4682.2 1690.81  4689.8 1690.40  4731.1 1689.86  4751.7 1689.89  4763.5 1689.75
  4799.0 1689.92  4804.2 1689.56  4839.7 1689.92  4915.8 1690.09  4921.0 1689.91
  4956.5 1689.93  4961.7 1689.76  4979.0 1689.94  4989.3 1689.81  4998.2 1689.47
  4998.5 1688.97  5002.0 1688.97  5002.2 1689.47  5010.2 1689.64  5033.8 1689.68
  5052.4 1690.27  5073.5 1691.52  5091.2 1692.00  5122.5 1692.24  5195.3 1693.49
#Mann=4,-1,0
  4622.9   0.075       0  4628.1    0.05       0  4998.2    0.05       0
  5002.2    0.05       0
Bank Sta=4998.2,5002.2
Exp/Cntr=0.3,0.1

Type RM Length L Ch R = 1,4223,237,237,237
BEGIN DESCRIPTION:
Elm 02 31 4222.66
END DESCRIPTION:
XS GIS Cut Line= 3
      1601435.08      6860155.99      1601639.04      6860307.88
      1601996.18      6860513.50
#Sta/Elev= 30
  4748.3 1693.34  4778.1 1693.02  4785.6 1693.20  4798.9 1691.93  4813.5 1692.02
  4821.9 1692.84  4846.3 1693.06  4885.3 1692.07  4907.4 1691.05  4913.6 1690.47
  4935.2 1689.32  4972.0 1688.47  4976.2 1687.79  4976.5 1687.29  4980.1 1687.29
  4980.3 1687.79  4992.9 1688.22  4998.5 1688.79  5014.1 1689.06  5021.0 1688.89
  5110.3 1689.71  5169.2 1689.84  5196.6 1690.34  5212.3 1690.21  5240.3 1690.87
  5292.8 1691.43  5321.0 1692.19  5330.2 1692.15  5373.3 1693.07  5414.7 1693.59
#Mann=4,-1,0
  4748.3   0.075       0  4846.3    0.05       0  4976.2    0.05       0
  4980.3    0.05       0
Bank Sta=4976.2,4980.3
Exp/Cntr=0.3,0.1

Type RM Length L Ch R = 1,3986,156,156,156
BEGIN DESCRIPTION:
Elm 02 31 3985.59
END DESCRIPTION:
XS GIS Cut Line= 3
      1601150.76      6860342.60      1601471.94      6860474.98
      1601866.87      6860722.35
#Sta/Elev= 30
  4655.5 1692.05  4670.9 1692.44  4685.0 1691.91  4703.3 1692.24  4768.2 1691.87
  4779.1 1691.70  4786.1 1690.53  4800.7 1689.85  4815.5 1689.92  4839.4 1692.43
  4876.4 1692.43  4898.1 1691.64  4908.9 1690.30  4916.6 1688.73  4922.0 1688.35
  4984.6 1688.05  4993.8 1687.81  4999.2 1687.05  5001.8 1686.19  5013.1 1686.07
  5013.3 1685.57  5017.0 1685.57  5017.3 1686.07  5036.4 1687.81  5057.6 1687.73
  5124.5 1690.37  5282.8 1691.52  5319.3 1692.31  5377.1 1692.56  5468.9 1693.77
#Mann=3,-1,0
  4655.5    0.05       0  5013.1    0.03       0  5017.3    0.05       0
Bank Sta=5013.1,5017.3
Exp/Cntr=0.3,0.1

Type RM Length L Ch R = 1,3830,205,205,205
BEGIN DESCRIPTION:
Elm 02 31 3829.92
END DESCRIPTION:
XS GIS Cut Line= 4
      1601342.12      6860445.98      1601392.32      6860506.73
      1601389.25      6860606.19      1601746.26      6861134.57
#Sta/Elev= 30
  4826.7 1692.31  4866.1 1691.49  4880.4 1690.38  4886.9 1688.47  4901.3 1688.07
  4903.7 1687.37  4981.3 1686.60  5007.7 1685.39  5007.9 1684.89  5011.6 1684.89
  5011.9 1685.39  5060.7 1687.94  5111.7 1688.63  5132.7 1689.59  5153.7 1689.23
  5162.6 1687.72  5168.6 1688.18  5176.2 1686.49  5183.6 1686.16  5240.6 1686.21
  5306.4 1686.99  5312.5 1688.45  5327.4 1687.83  5333.5 1689.15  5342.4 1688.86
  5348.4 1689.55  5378.4 1689.58  5384.4 1690.71  5399.4 1691.26  5642.7 1692.68
#Mann=3,-1,0
  4826.7    0.05       0  5007.7    0.03       0  5011.9    0.05       0
Bank Sta=5007.7,5011.9
Exp/Cntr=0.3,0.1

Type RM Length L Ch R = 1,3625,599,599,599
BEGIN DESCRIPTION:
Elm 02 31 3624.84
END DESCRIPTION:
XS GIS Cut Line= 4
      1601213.47      6860462.98      1601239.51      6860740.31
      1601270.78      6860971.09      1601337.60      6861293.71
#Sta/Elev= 30
  4724.6 1688.42  4759.8 1688.66  4830.1 1687.17  4903.4 1686.72  4930.5 1687.91
  4940.6 1686.66  4960.6 1687.11  4970.7 1686.24  4978.6 1683.63  4978.9 1683.13
  4982.6 1683.13  4982.9 1683.63  5003.1 1683.68  5011.4 1685.29  5051.3 1685.04
  5071.5 1685.37  5083.9 1686.45  5142.1 1685.83  5156.5 1686.33  5202.6 1685.14
  5222.8 1685.20  5233.1 1685.92  5280.2 1685.22  5285.3 1685.86  5330.3 1685.99
  5345.2 1686.90  5406.5 1686.05  5425.6 1686.33  5430.7 1687.62  5565.5 1688.46
#Mann=3,-1,0
  4724.6    0.05       0  4978.6    0.03       0  4982.9    0.05       0
Bank Sta=4978.6,4982.9
Exp/Cntr=0.3,0.1

Type RM Length L Ch R = 1,3026,285,285,285
BEGIN DESCRIPTION:
Elm 02 31 3026.32
END DESCRIPTION:
XS GIS Cut Line= 3
      1601022.53      6860991.68      1601135.38      6861208.70
      1601243.87      6861466.92
#Sta/Elev= 30
  4756.4 1685.95  4776.5 1685.90  4786.1 1686.42  4808.6 1686.61  4859.3 1686.64
  4897.9 1685.77  4920.0 1684.87  4925.6 1685.00  4932.6 1682.03  4942.1 1681.40
  4964.2 1680.90  4969.9 1681.15  4977.7 1680.89  4984.2 1680.33  4984.5 1679.83
  4988.2 1679.83  4988.5 1680.33  4997.8 1680.91  5062.2 1681.41  5067.7 1681.77
  5086.0 1681.87  5091.4 1682.27  5115.2 1682.45  5120.6 1683.10  5162.7 1683.95
  5173.8 1684.45  5215.6 1684.82  5221.0 1685.13  5274.0 1684.20  5281.1 1683.76
#Mann=3,-1,0
  4756.4    0.05       0  4984.2    0.03       0  4988.5    0.05       0
Bank Sta=4984.2,4988.5
Exp/Cntr=0.3,0.1

Type RM Length L Ch R = 1,2741,109,109,109
BEGIN DESCRIPTION:
Elm 02 31 2740.73
END DESCRIPTION:
XS GIS Cut Line= 3
      1600916.19      6860990.58      1600901.00      6861339.99
      1600893.41      6861609.04
#Sta/Elev= 30
  4651.8 1684.50  4699.3 1684.47  4709.3 1685.50  4729.3 1685.66  4759.3 1685.33
  4789.4 1685.30  4799.4 1684.92  4809.4 1682.38  4819.4 1680.41  4839.4 1679.10
  4849.4 1678.72  4869.4 1678.46  4899.5 1678.46  4929.5 1677.74  4949.5 1677.62
  4969.5 1677.09  5027.3 1676.38  5027.6 1675.88  5031.6 1675.88  5031.9 1676.38
  5035.8 1676.38  5040.8 1676.76  5069.6 1676.52  5129.6 1677.41  5149.6 1678.70
  5209.6 1680.79  5239.6 1682.94  5249.6 1683.20  5259.7 1683.94  5270.7 1684.34
#Mann=3,-1,0
  4651.8    0.05       0  5027.3    0.05       0  5031.9    0.05       0
Bank Sta=5027.3,5031.9
Exp/Cntr=0.3,0.1

Type RM Length L Ch R = 1,2632,274,274,274
BEGIN DESCRIPTION:
Elm 02 31 2632.17
END DESCRIPTION:
XS GIS Cut Line= 3
      1600793.58      6860977.58      1600792.50      6861341.08
      1600763.25      6861633.52
#Sta/Elev= 30
  4639.1 1684.92  4699.5 1683.81  4709.5 1684.57  4729.5 1685.03  4799.5 1684.13
  4809.5 1683.09  4819.5 1681.00  4879.5 1677.80  4909.5 1675.57  4929.5 1675.18
  4943.4 1674.23  4947.2 1673.95  4947.5 1673.45  4951.5 1673.45  4951.8 1673.95
  4979.5 1674.48  5049.8 1673.98  5079.9 1674.24  5090.0 1674.57  5098.6 1675.71
  5110.1 1677.08  5120.1 1677.57  5126.7 1678.50  5140.2 1679.13  5150.3 1680.42
  5232.2 1683.44  5250.8 1683.69  5270.9 1684.44  5280.9 1685.24  5296.5 1685.57
#Mann=5,-1,0
  4639.1    0.05       0  4943.4   0.075       0  4947.2    0.07       0
  4951.8   0.075       0  5098.6    0.05       0
Bank Sta=4947.2,4951.8
Exp/Cntr=0.3,0.1

Type RM Length L Ch R = 1,2358,317,317,317
BEGIN DESCRIPTION:
Elm 02 31 2358.04
END DESCRIPTION:
XS GIS Cut Line= 3
      1600587.86      6861003.80      1600555.31      6861234.27
      1600517.55      6861619.67
#Sta/Elev= 30
  4768.9 1682.83  4821.9 1682.02  4826.9 1681.63  4843.8 1681.58  4853.9 1680.87
  4874.1 1678.71  4885.2 1678.09  4893.0 1677.58  4903.5 1676.18  4914.5 1675.16
  4934.7 1673.91  5043.2 1673.83  5043.6 1673.33  5047.6 1673.33  5047.9 1673.83
  5053.4 1674.91  5058.4 1675.35  5075.7 1676.04  5095.8 1677.49  5112.8 1679.33
  5126.0 1680.59  5146.1 1681.79  5154.9 1683.10  5159.9 1682.30  5166.2 1682.35
  5186.3 1683.23  5261.4 1684.42  5266.6 1684.82  5276.7 1684.58  5388.9 1685.69
#Mann=6,-1,0
  4768.9    0.05       0  4885.2   0.075       0  4903.5    0.12       0
  5043.2    0.07       0  5047.9    0.12       0  5112.8    0.05       0
Bank Sta=5043.2,5047.9
Exp/Cntr=0.3,0.1

Type RM Length L Ch R = 1,2041,84,84,84
BEGIN DESCRIPTION:
Elm 02 31 2040.77
END DESCRIPTION:
XS GIS Cut Line= 3
      1600249.19      6861103.41      1600321.88      6861370.31
      1600372.87      6861648.05
#Sta/Elev= 30
  4723.4 1683.13  4769.7 1682.51  4799.1 1681.78  4804.2 1682.13  4811.1 1682.14
  4873.3 1681.29  4878.6 1680.86  4894.0 1680.88  4904.4 1680.09  4913.1 1678.61
  4918.3 1678.41  4925.1 1675.96  4935.4 1674.03  4979.2 1673.89  5005.5 1673.83
  5005.8 1673.33  5009.9 1673.33  5010.2 1673.83  5044.2 1674.58  5064.3 1674.57
  5097.3 1674.59  5150.2 1674.15  5170.5 1677.50  5190.8 1681.58  5208.6 1682.70
  5213.7 1682.53  5241.7 1683.86  5251.9 1684.14  5261.7 1683.89  5282.4 1684.26
#Mann=5,-1,0
  4723.4    0.05       0  4979.2    0.12       0  5005.5    0.07       0
  5010.2    0.12       0  5064.3    0.05       0
Bank Sta=5005.5,5010.2
Exp/Cntr=0.3,0.1

Type RM Length L Ch R = 1,1957,293,293,293
BEGIN DESCRIPTION:
Elm 02 31 1957.46
END DESCRIPTION:
XS GIS Cut Line= 3
      1600108.13      6861103.39      1600244.84      6861390.92
      1600290.20      6861660.96
#Sta/Elev= 30
  4684.4 1683.86  4737.3 1683.03  4754.5 1681.23  4760.1 1681.07  4777.2 1678.63
  4782.8 1678.68  4789.2 1677.15  4799.9 1675.60  4805.5 1675.80  4811.3 1674.77
  4828.2 1673.15  4833.7 1673.47  4844.5 1672.80  4850.9 1671.80  4856.5 1672.71
  4873.6 1670.89  5068.4 1670.83  5068.7 1670.33  5072.8 1670.33  5073.2 1670.83
  5141.8 1671.11  5155.8 1672.31  5162.1 1674.49  5172.2 1676.80  5182.3 1679.75
  5192.5 1681.51  5202.6 1682.31  5216.4 1682.47  5233.0 1683.52  5276.6 1683.76
#Mann=3,-1,0
  4684.4    0.05       0  5068.4    0.05       0  5073.2    0.05       0
Bank Sta=5068.4,5073.2
Exp/Cntr=0.3,0.1

Type RM Length L Ch R = 1,1664,227,227,227
BEGIN DESCRIPTION:
Elm 02 31 1664.27
END DESCRIPTION:
XS GIS Cut Line= 3
      1599883.50      6861144.59      1599951.87      6861395.26
      1600092.94      6861732.74
#Sta/Elev= 30
  4741.0 1684.23  4802.6 1683.69  4837.2 1681.75  4842.4 1681.14  4848.2 1679.58
  4882.1 1673.52  4889.7 1671.77  4900.0 1671.10  5047.8 1670.86  5048.2 1670.36
  5052.3 1670.36  5052.6 1670.86  5112.2 1670.88  5150.8 1671.38  5156.3 1673.01
  5174.6 1673.71  5180.1 1675.19  5198.4 1676.73  5203.9 1678.15  5220.6 1678.88
  5233.1 1679.98  5251.5 1680.99  5274.8 1680.91  5286.1 1681.81  5304.5 1682.09
  5318.1 1682.70  5328.3 1682.60  5333.7 1683.31  5339.8 1682.85  5366.6 1682.53
#Mann=3,-1,0
  4741.0    0.05       0  5047.8    0.05       0  5052.6    0.05       0
Bank Sta=5047.8,5052.6
Exp/Cntr=0.3,0.1

Type RM Length L Ch R = 1,1437,43,43,43
BEGIN DESCRIPTION:
Elm 02 31 1436.86
END DESCRIPTION:
XS GIS Cut Line= 5
      1599807.55      6861222.70      1599821.01      6861572.17
      1599847.70      6861639.40      1599910.15      6861770.36
      1600009.35      6861878.09
#Sta/Elev= 30
  4650.7 1683.73  4686.0 1683.67  4717.7 1682.30  4766.1 1681.26  4786.1 1679.61
  4806.1 1677.19  4836.1 1674.34  4866.2 1672.41  4876.2 1671.37  4896.2 1670.94
  4970.3 1670.88  4970.7 1670.38  4974.8 1670.38  4975.1 1670.88  5039.0 1670.99
  5060.5 1671.48  5128.4 1671.34  5145.5 1671.99  5151.1 1671.65  5168.2 1673.17
  5173.7 1672.25  5190.9 1672.88  5213.6 1674.97  5217.7 1676.20  5233.7 1678.87
  5241.1 1678.90  5269.0 1680.46  5276.2 1680.25  5325.6 1681.46  5364.3 1682.90
#Mann=3,-1,0
  4650.7    0.05       0  4970.3    0.05       0  4975.1    0.05       0
Bank Sta=4970.3,4975.1
Exp/Cntr=0.3,0.1

Type RM Length L Ch R = 1,1394,98,98,98
BEGIN DESCRIPTION:
Elm 02 31 1394.29
END DESCRIPTION:
XS GIS Cut Line= 4
      1599752.22      6861279.18      1599791.28      6861602.51
      1599815.15      6861719.70      1599957.28      6861878.10
#Sta/Elev= 30
  4674.6 1683.33  4683.5 1683.72  4764.1 1681.86  4814.4 1681.94  4864.8 1676.72
  4903.1 1676.59  4908.2 1673.98  4955.5 1676.13  4965.5 1676.22  4985.1 1675.11
  4990.2 1676.05  5000.3 1676.11  5026.3 1675.27  5042.8 1673.27  5047.9 1675.43
  5093.4 1674.01  5098.5 1675.30  5125.7 1675.18  5146.7 1674.27  5154.1 1673.37
  5180.1 1672.59  5180.5 1672.09  5184.6 1672.09  5184.9 1672.59  5196.8 1673.02
  5211.0 1675.06  5217.7 1675.21  5225.1 1676.81  5238.6 1678.40  5332.7 1682.31
#Mann=3,-1,0
  4674.6    0.05       0  5180.1    0.05       0  5184.9    0.05       0
Bank Sta=5180.1,5184.9
Exp/Cntr=0.3,0.1

Type RM Length L Ch R = 1,1296,97,97,97
BEGIN DESCRIPTION:
Elm 02 31 1295.95
END DESCRIPTION:
XS GIS Cut Line= 4
      1599639.36      6861346.41      1599749.83      6861688.49
      1599783.08      6861788.26      1599930.65      6861891.80
#Sta/Elev= 30
  4641.7 1683.33  4742.3 1682.12  4838.4 1680.06  4864.0 1677.93  4875.7 1675.04
  4895.6 1672.43  4907.7 1669.62  4934.5 1666.42  4979.6 1661.72  4990.1 1660.98
  5001.2 1661.17  5027.8 1658.52  5028.1 1658.02  5032.2 1658.02  5032.6 1658.52
  5035.4 1659.60  5061.8 1660.24  5067.1 1661.16  5093.4 1661.29  5098.7 1663.89
  5103.6 1663.17  5120.9 1663.89  5129.5 1668.65  5135.6 1668.97  5150.4 1672.81
  5165.2 1674.06  5171.3 1676.01  5221.9 1680.20  5257.6 1681.69  5286.6 1681.87
#Mann=3,-1,0
  4641.7    0.05       0  5027.8    0.05       0  5032.6    0.05       0
Bank Sta=5027.8,5032.6
Exp/Cntr=0.3,0.1

Type RM Length L Ch R = 1,1199,181,181,181
BEGIN DESCRIPTION:
Elm 02 31 1198.81
END DESCRIPTION:
XS GIS Cut Line= 4
      1599461.63      6861500.90      1599685.77      6861759.67
      1599776.74      6861844.74      1599926.92      6861908.11
#Sta/Elev= 30
  4658.0 1680.85  4680.0 1681.32  4729.4 1680.30  4772.2 1680.60  4842.4 1678.91
  4870.9 1675.50  4899.4 1669.20  4942.2 1662.60  4963.0 1660.38  4984.9 1659.78
  4995.9 1657.36  5002.8 1657.36  5005.7 1656.25  5017.5 1655.68  5017.8 1655.18
  5021.9 1655.18  5022.3 1655.68  5040.9 1656.16  5048.2 1658.01  5069.2 1660.44
  5090.7 1665.47  5097.5 1666.25  5111.7 1669.33  5123.6 1672.93  5148.1 1675.75
  5166.4 1676.56  5177.3 1678.23  5195.6 1679.53  5231.6 1681.20  5287.9 1681.92
#Mann=3,-1,0
  4658.0    0.05       0  5017.5    0.05       0  5022.3    0.05       0
Bank Sta=5017.5,5022.3
Exp/Cntr=0.3,0.1

Type RM Length L Ch R = 1,1018,263,263,263
BEGIN DESCRIPTION:
Elm 02 31 1017.8
END DESCRIPTION:
XS GIS Cut Line= 4
      1598736.86      6861344.71      1599335.79      6861885.05
      1599588.82      6861905.71      1599854.10      6861920.30
#Sta/Elev= 30
  3939.6 1674.24  3962.1 1672.05  3983.0 1668.04  3990.5 1665.78  4011.4 1663.93
  4039.8 1663.21  4046.6 1663.66  4223.7 1662.58  4372.4 1663.03  4577.9 1660.99
  4684.0 1660.76  4825.7 1658.33  4926.1 1659.32  4976.2 1658.62  4986.3 1657.28
  5003.9 1656.36  5004.3 1655.86  5008.4 1655.86  5008.7 1656.36  5026.3 1657.06
  5046.4 1659.68  5096.4 1663.92  5126.5 1667.92  5137.2 1670.85  5146.5 1672.58
  5156.5 1673.56  5166.6 1674.42  5196.6 1675.07  5226.6 1679.11  5265.8 1681.04
#Mann=3,-1,0
  3939.6    0.05       0  5003.9    0.05       0  5008.7    0.05       0
Bank Sta=5003.9,5008.7
Exp/Cntr=0.3,0.1

Type RM Length L Ch R = 1,755,180,180,180
BEGIN DESCRIPTION:
Elm 02 31 754.6
END DESCRIPTION:
XS GIS Cut Line= 3
      1598697.73      6861609.41      1599499.59      6862141.48
      1599686.20      6862277.75
#Sta/Elev= 30
  4039.0 1662.95  4461.6 1661.57  4491.7 1660.12  4599.8 1659.48  4656.2 1660.41
  4750.3 1660.02  4779.8 1661.86  4826.1 1653.58  4826.5 1653.08  4831.0 1653.58
  4851.8 1654.85  4864.6 1659.01  4900.7 1661.17  4972.9 1660.36  4987.9 1657.40
  4995.6 1654.47  5001.3 1654.47  5017.5 1657.78  5067.7 1661.60  5088.6 1666.55
  5094.8 1666.21  5103.3 1669.57  5109.5 1668.66  5117.9 1671.43  5124.1 1671.11
  5138.8 1676.47  5145.0 1676.16  5153.5 1679.01  5195.2 1681.16  5232.4 1680.04
#Mann=4,-1,0
  4039.0    0.05       0  4656.2    0.12       0  4826.1    0.07       0
  4831.0    0.12       0
Bank Sta=4826.1,4831
Exp/Cntr=0.3,0.1

Type RM Length L Ch R = 1,575,193,193,193
BEGIN DESCRIPTION:
Elm 02 31 575.23
END DESCRIPTION:
XS GIS Cut Line= 3
      1598706.48      6861876.38      1599404.57      6862287.92
      1599554.54      6862378.18
#Sta/Elev= 30
  4189.7 1662.65  4262.6 1661.15  4292.5 1661.74  4518.3 1660.89  4709.5 1658.36
  4774.0 1658.77  4811.1 1657.84  4816.9 1657.95  4832.5 1660.79  4869.6 1661.35
  4875.5 1660.29  4896.9 1660.17  4912.6 1655.91  4919.3 1652.86  4925.7 1652.38
  4926.1 1651.88  4930.7 1652.38  4942.5 1652.81  4955.5 1656.58  4986.8 1659.08
  5003.2 1657.58  5008.2 1654.16  5014.0 1652.63  5023.7 1653.29  5035.6 1656.78
  5082.9 1666.12  5124.7 1676.66  5161.6 1680.86  5171.2 1681.16  5175.1 1681.28
#Mann=6,-1,0
  4189.7    0.05       0  4709.5    0.12       0  4925.7    0.07       0
  4930.7    0.12       0  5082.9    0.05       0  5171.2    0.12       0
Bank Sta=4925.7,4930.7
Exp/Cntr=0.3,0.1

Type RM Length L Ch R = 1,382,201,201,201
BEGIN DESCRIPTION:
Elm 02 31 381.8
END DESCRIPTION:
XS GIS Cut Line= 4
      1598697.78      6861971.86      1599197.75      6862385.39
      1599301.21      6862444.39      1599499.79      6862575.69
#Sta/Elev= 30
  4234.0 1662.05  4314.5 1660.99  4520.3 1660.93  4555.5 1660.34  4592.0 1661.09
  4705.3 1660.61  4726.1 1661.00  4789.9 1660.50  4868.1 1659.04  4897.6 1661.06
  4903.3 1660.70  4940.8 1661.91  4948.7 1661.51  4956.6 1660.02  4978.2 1652.55
  4984.0 1651.16  4999.4 1649.91  4999.8 1649.41  5004.0 1649.41  5004.4 1649.91
  5021.0 1650.73  5051.1 1658.87  5078.4 1662.98  5114.4 1671.14  5123.3 1672.18
  5129.3 1674.04  5150.4 1677.30  5165.5 1678.84  5186.5 1679.72  5240.0 1680.00
#Mann=3,-1,0
  4234.0    0.05       0  4999.4    0.05       0  5004.4    0.05       0
Bank Sta=4999.4,5004.4
Exp/Cntr=0.3,0.1

Type RM Length L Ch R = 1,181,89,89,89
BEGIN DESCRIPTION:
Elm 02 31 180.98
END DESCRIPTION:
XS GIS Cut Line= 3
      1598697.78      6862080.37      1599168.54      6862576.12
      1599389.90      6862701.99
#Sta/Elev= 30
  4316.8 1661.63  4362.7 1660.55  4631.3 1660.41  4695.2 1659.38  4730.4 1660.52
  4787.0 1660.51  4886.1 1659.15  4935.5 1661.27  4938.8 1660.64  4963.8 1657.85
  4985.2 1654.31  4992.1 1652.25  5000.5 1652.31  5014.0 1648.53  5019.8 1649.07
  5029.9 1647.76  5035.6 1648.46  5049.0 1647.08  5049.4 1646.58  5054.0 1647.08
  5082.1 1649.24  5116.4 1655.23  5122.9 1657.62  5138.0 1660.04  5153.8 1664.56
  5181.2 1670.63  5197.1 1672.79  5203.4 1674.95  5226.5 1677.39  5255.1 1678.08
#Mann=5,-1,0
  4316.8    0.05       0  4938.8    0.12       0  5049.0    0.07       0
  5054.0    0.12       0  5082.1    0.05       0
Bank Sta=5049,5054
Exp/Cntr=0.3,0.1

Type RM Length L Ch R = 1,92,76,76,76
BEGIN DESCRIPTION:
Elm 02 31 91.56
END DESCRIPTION:
XS GIS Cut Line= 5
      1598695.60      6862197.55      1598938.83      6862561.75
      1599136.43      6862656.85      1599198.06      6862702.85
      1599399.47      6862781.85
#Sta/Elev= 30
  4343.6 1661.22  4407.9 1659.46  4711.3 1656.93  4798.7 1657.26  4866.1 1656.88
  4879.7 1652.99  4885.8 1652.77  4886.2 1652.27  4890.8 1652.77  4896.8 1655.85
  4910.5 1658.06  4954.9 1657.37  4977.1 1654.09  4992.8 1654.83  4997.3 1657.14
  5008.2 1658.34  5029.0 1657.15  5043.6 1657.98  5049.9 1655.63  5064.5 1654.21
  5108.8 1654.89  5127.9 1656.87  5130.3 1656.18  5133.2 1655.35  5138.9 1658.09
  5163.0 1662.92  5187.5 1670.51  5211.9 1676.17  5241.7 1678.42  5294.1 1679.30
#Mann=5,-1,0
  4343.6    0.05       0  4798.7    0.12       0  4885.8    0.07       0
  4890.8    0.12       0  5130.3    0.05       0
Bank Sta=4885.8,4890.8
Exp/Cntr=0.3,0.1

Type RM Length L Ch R = 1,16,0,0,0
BEGIN DESCRIPTION:
Elm 02 31 976.764
END DESCRIPTION:
XS GIS Cut Line= 4
      1598695.62      6862267.03      1598868.27      6862596.45
      1599105.05      6862721.95      1599395.34      6862861.52
#Sta/Elev= 30
  4360.1 1660.62  4478.5 1658.62  4827.1 1656.79  4833.6 1655.47  4850.0 1657.01
  4864.1 1656.24  4877.6 1648.99  4894.0 1652.39  4899.6 1649.79  4915.9 1652.48
  4921.6 1648.40  4937.9 1652.02  4943.6 1649.17  4954.3 1650.21  4966.0 1647.61
  5000.0 1647.48  5004.0 1651.25  5021.0 1648.42  5026.6 1651.42  5043.7 1648.44
  5046.9 1646.54  5047.9 1646.04  5096.8 1646.54  5100.0 1654.60  5133.1 1654.23
  5155.4 1658.19  5190.6 1666.48  5207.7 1672.48  5230.3 1677.03  5322.1 1678.92
#Mann=5,-1,0
  4360.1    0.05       0  4827.1    0.12       0  5046.9    0.07       0
  5096.8    0.12       0  5155.4    0.05       0
Bank Sta=5046.9,5096.8
Exp/Cntr=0.3,0.1

Chan Stop Cuts=-1
