--- Elm 46.prj (project) ---

Proj Title=Elm 46 Base Level Engineering
Current Plan=p01
Default Exp/Contr=0.3,0.1
English Units
Geom File=g01
Flow File=f01
Plan File=p01
BEGIN DESCRIPTION:
Elm 46
END DESCRIPTION:

--- Elm 46.p01 (plan) ---

Plan Title=Multiple Run
Short Identifier=Multiple
Geom File=g01
Flow File=f01
Subcritical Flow
K Sum by GR= 0
Std Step Tol= 0.01
Critical Tol= 0.01
Num of Std Step Trials= 20
Max Error Tol= 0.3
Flow Tol Ratio= 0.001
Split Flow NTrial= 30
Split Flow Tol= 0.02
Split Flow Ratio= 0.02
Log Output Level= 0
Friction Slope Method= 1
Unsteady Friction Slope Method= 2
Unsteady Bridges Friction Slope Method= 1
Parabolic Critical Depth
Global Vel Dist=  1 , 1 , 1
Global Log Level= 0
CheckData=True
Encroach Param= -1, 0, 0, 0
BEGIN DESCRIPTION:
Multiple Run
END DESCRIPTION:

--- Elm 46.f01 (steady flow) ---

Flow Title=Multiple
Number of Profiles=7
Profile Names=10-year,25-year,50-year,1pct_min,100-year,1pct_plu,500-year
River Rch & RM= Elm 46,Reach-1,3430
     151     207     255     195     313     430     476
Boundary for River Rch & Prof#=Elm 46,Reach-1,1
Up Type=0
Dn Type=3
Dn Slope=0.005
Boundary for River Rch & Prof#=Elm 46,Reach-1,2
Up Type=0
Dn Type=3
Dn Slope=0.005
Boundary for River Rch & Prof#=Elm 46,Reach-1,3
Up Type=0
Dn Type=3
Dn Slope=0.005
Boundary for River Rch & Prof#=Elm 46,Reach-1,4
Up Type=0
Dn Type=3
Dn Slope=0.005
Boundary for River Rch & Prof#=Elm 46,Reach-1,5
Up Type=0
Dn Type=3
Dn Slope=0.005
Boundary for River Rch & Prof#=Elm 46,Reach-1,6
Up Type=0
Dn Type=3
Dn Slope=0.005
Boundary for River Rch & Prof#=Elm 46,Reach-1,7
Up Type=0
Dn Type=3
Dn Slope=0.005

--- Elm 46.g01 (geometry) ---

Geom Title=Existing Conditions

River Reach=Elm 46,Reach-1
Reach XY= 30
      1511605.00      6771788.00      1511660.79      6771836.09
      1511811.19      6771845.81      1512025.39      6772057.84
      1512115.77      6772247.68      1512244.22      6772378.32
      1512268.63      6772451.21      1512447.14      6772631.83
      1512458.83      6772736.41      1512552.67      6772893.97
      1512558.62      6772986.50      1512646.86      6773081.96
      1512696.96      6773184.68      1512657.36      6773243.90
      1512655.95      6773327.51      1512751.44      6773439.47
      1512758.76      6773586.44      1512877.81      6773811.95
      1512910.71      6773835.92      1513003.78      6773841.53
      1513047.63      6773881.63      1513054.13      6773927.31
      1513012.91      6773984.77      1513021.30      6774004.70
      1513145.34      6774127.83      1513194.51      6774137.52
      1513244.35      6774098.11      1513263.15      6774031.96
      1513334.86      6773957.76      1513405.00      6773938.00

Type RM Length L Ch R = 1,3430,22,22,22
BEGIN DESCRIPTION:
elmc399
END DESCRIPTION:
XS GIS Cut Line= 3
      1511605.02      6771887.96      1511641.50      6771825.08
      1511754.98      6771588.04
#Sta/Elev= 30
  4927.3 2268.08  4930.1 2268.08  4935.1 2264.01  4940.9 2264.87  4950.4 2257.64
  4956.7 2257.17  4962.4 2253.26  4972.4 2252.83  4978.2 2249.78  5020.1 2242.50
  5020.3 2242.00  5023.8 2242.00  5024.1 2242.50  5030.0 2245.54  5039.2 2249.39
  5052.2 2252.62  5061.9 2254.17  5067.4 2254.14  5074.4 2255.88  5096.5 2259.42
  5112.7 2261.12  5129.8 2263.56  5158.1 2269.10  5174.2 2271.03  5180.7 2272.45
  5218.5 2276.68  5248.7 2282.67  5254.3 2283.25  5260.1 2285.00  5262.8 2285.00
#Mann=3,-1,0
  4927.3    0.16       0  5020.1    0.07       0  5024.1    0.16       0
Bank Sta=5020.1,5024.1
Exp/Cntr=0.3,0.1

Type RM Length L Ch R = 1,3408,35,35,35
BEGIN DESCRIPTION:
elmc554
END DESCRIPTION:
XS GIS Cut Line= 3
      1511636.40      6771908.55      1511661.36      6771835.84
      1511752.50      6771688.29
#Sta/Elev= 30
  4923.4 2273.25  4926.3 2273.25  4931.9 2271.14  4937.2 2270.13  4955.7 2263.09
  4963.1 2256.72  4976.8 2250.65  4994.4 2245.46  5016.0 2243.62  5019.9 2241.88
  5020.2 2241.38  5023.7 2241.38  5023.9 2241.88  5031.4 2244.30  5037.3 2247.64
  5052.7 2252.13  5058.6 2251.82  5068.1 2253.23  5074.0 2252.63  5080.0 2254.21
  5089.4 2255.98  5095.2 2255.29  5110.6 2259.23  5116.5 2258.55  5126.0 2261.45
  5131.9 2262.59  5147.3 2266.70  5162.3 2268.90  5171.3 2271.24  5173.7 2271.24
#Mann=3,-1,0
  4923.4    0.16       0  5019.9    0.07       0  5023.9    0.16       0
Bank Sta=5019.9,5023.9
Exp/Cntr=0.3,0.1

Type RM Length L Ch R = 1,3373,22,22,22
BEGIN DESCRIPTION:
elmc557
END DESCRIPTION:
XS GIS Cut Line= 3
      1511673.30      6771930.25      1511696.09      6771833.67
      1511758.47      6771691.70
#Sta/Elev= 30
  4903.8 2273.11  4907.5 2273.11  4926.7 2268.97  4932.4 2265.10  4947.2 2257.79
  4957.5 2253.35  4967.8 2247.93  4986.3 2240.84  4986.6 2240.34  4990.1 2240.34
  4990.3 2240.84  4998.2 2242.76  5003.0 2242.76  5008.3 2243.54  5013.7 2243.78
  5031.1 2246.80  5037.1 2249.48  5052.9 2250.72  5060.4 2251.79  5065.9 2252.03
  5083.8 2255.34  5089.2 2255.77  5096.6 2258.10  5107.1 2260.35  5112.6 2260.61
  5118.4 2263.05  5129.4 2265.58  5135.9 2267.72  5151.2 2269.52  5158.1 2271.24
#Mann=3,-1,0
  4903.8    0.16       0  4986.3    0.07       0  4990.3    0.16       0
Bank Sta=4986.3,4990.3
Exp/Cntr=0.3,0.1

Type RM Length L Ch R = 1,3351,29,29,29
BEGIN DESCRIPTION:
elmc555
END DESCRIPTION:
XS GIS Cut Line= 3
      1511700.42      6771910.72      1511716.70      6771840.18
      1511768.78      6771687.19
#Sta/Elev= 30
  4924.2 2263.36  4928.2 2263.36  4937.3 2258.85  4957.8 2250.98  4964.8 2245.65
  4970.0 2245.63  4976.3 2241.01  4976.6 2240.51  4980.1 2240.51  4980.3 2241.01
  4988.6 2241.40  4995.1 2242.49  5005.5 2242.97  5010.8 2242.33  5020.0 2244.29
  5030.6 2247.84  5036.9 2251.04  5042.1 2251.11  5051.7 2253.24  5062.3 2253.16
  5068.2 2253.95  5073.5 2255.20  5094.0 2258.30  5099.6 2260.61  5104.9 2260.87
  5115.1 2263.23  5125.7 2266.33  5130.9 2268.45  5155.1 2271.41  5158.2 2271.41
#Mann=3,-1,0
  4924.2    0.16       0  4976.3    0.07       0  4980.3    0.16       0
Bank Sta=4976.3,4980.3
Exp/Cntr=0.3,0.1

Type RM Length L Ch R = 1,3322,26,26,26
BEGIN DESCRIPTION:
elmc558
END DESCRIPTION:
XS GIS Cut Line= 3
      1511724.31      6771924.77      1511747.08      6771835.84
      1511791.57      6771705.63
#Sta/Elev= 30
  4909.8 2267.06  4916.8 2265.58  4927.1 2262.28  4932.5 2258.87  4937.7 2258.43
  4947.8 2253.99  4958.1 2250.26  4968.1 2245.35  4973.3 2244.97  4978.7 2240.31
  4987.0 2239.45  4987.3 2238.95  4990.8 2238.95  4991.0 2239.45  4997.9 2240.84
  5001.6 2240.84  5007.6 2241.57  5012.9 2241.86  5038.9 2251.68  5044.2 2250.30
  5052.2 2252.41  5062.7 2254.33  5070.2 2256.60  5075.5 2256.33  5083.9 2259.42
  5094.4 2261.27  5101.6 2263.26  5115.6 2266.37  5132.9 2269.67  5139.2 2269.85
#Mann=3,-1,0
  4909.8    0.16       0  4987.0    0.07       0  4991.0    0.16       0
Bank Sta=4987,4991
Exp/Cntr=0.3,0.1

Type RM Length L Ch R = 1,3296,19,19,19
BEGIN DESCRIPTION:
elmc559
END DESCRIPTION:
XS GIS Cut Line= 3
      1511732.99      6771939.98      1511772.04      6771841.26
      1511817.62      6771694.75
#Sta/Elev= 30
  4890.2 2266.38  4893.9 2266.38  4903.1 2265.14  4914.2 2261.39  4956.9 2249.30
  4962.9 2244.90  4968.3 2243.60  4978.4 2240.17  4987.3 2239.10  4990.7 2237.33
  4990.9 2236.83  4994.4 2236.83  4994.7 2237.33  4995.4 2239.46  5000.7 2239.46
  5010.3 2241.72  5019.3 2244.33  5024.6 2243.66  5031.2 2246.73  5051.9 2251.23
  5057.1 2251.74  5062.6 2253.98  5083.6 2260.05  5089.6 2262.64  5104.5 2265.83
  5115.0 2267.38  5122.2 2268.96  5127.4 2268.90  5145.5 2270.78  5149.8 2270.78
#Mann=3,-1,0
  4890.2    0.16       0  4990.7    0.07       0  4994.7    0.16       0
Bank Sta=4990.7,4994.7
Exp/Cntr=0.3,0.1

Type RM Length L Ch R = 1,3277,17,17,17
BEGIN DESCRIPTION:
elmc560
END DESCRIPTION:
XS GIS Cut Line= 3
      1511738.39      6771944.37      1511791.57      6771839.09
      1511824.12      6771703.49
#Sta/Elev= 30
  4881.9 2268.05  4884.5 2266.38  4890.1 2264.69  4900.2 2263.12  4922.6 2257.18
  4929.0 2254.70  4945.1 2251.41  4951.3 2248.55  4956.9 2248.25  4967.5 2243.37
  4973.6 2238.80  4979.2 2238.56  4987.9 2236.58  4988.1 2236.08  4991.6 2236.08
  4991.9 2236.58  4995.9 2239.47  5003.0 2239.44  5021.5 2243.83  5031.3 2246.77
  5036.5 2246.89  5042.1 2249.35  5073.0 2257.96  5078.5 2261.14  5103.8 2266.27
  5114.1 2267.50  5120.4 2268.90  5125.6 2268.76  5134.4 2269.95  5139.3 2269.95
#Mann=3,-1,0
  4881.9    0.16       0  4987.9    0.07       0  4991.9    0.16       0
Bank Sta=4987.9,4991.9
Exp/Cntr=0.3,0.1

Type RM Length L Ch R = 1,3260,33,33,33
BEGIN DESCRIPTION:
elmc556
END DESCRIPTION:
XS GIS Cut Line= 3
      1511738.43      6771955.16      1511810.02      6771841.26
      1511845.52      6771691.74
#Sta/Elev= 30
  4869.1 2269.99  4871.9 2268.05  4877.8 2266.31  4887.2 2264.69  4893.1 2262.96
  4914.3 2257.92  4929.6 2254.71  4936.6 2252.58  4950.8 2249.72  4960.2 2247.05
  4966.1 2244.97  4972.0 2242.04  4981.4 2238.20  4987.3 2237.41  4993.7 2237.13
  4993.9 2236.63  4997.4 2236.63  4997.7 2237.13  5002.6 2240.53  5007.9 2240.67
  5017.3 2243.21  5027.5 2245.24  5037.8 2248.01  5044.9 2249.45  5050.0 2251.28
  5068.6 2255.99  5087.1 2262.39  5120.0 2267.68  5134.4 2269.08  5157.3 2271.97
#Mann=3,-1,0
  4869.1    0.16       0  4993.7    0.07       0  4997.7    0.16       0
Bank Sta=4993.7,4997.7
Exp/Cntr=0.3,0.1

Type RM Length L Ch R = 1,3227,41,41,41
BEGIN DESCRIPTION:
elmc561
END DESCRIPTION:
XS GIS Cut Line= 3
      1511759.04      6771962.76      1511834.98      6771861.88
      1511876.92      6771701.64
#Sta/Elev= 30
  4879.1 2266.33  4900.6 2260.35  4908.9 2258.98  4915.1 2256.51  4929.7 2254.07
  4936.0 2251.36  4944.3 2250.70  4950.5 2248.26  4958.9 2246.15  4965.1 2236.93
  4979.7 2230.06  4986.0 2216.10  4994.3 2205.14  4998.5 2204.83  4998.8 2204.33
  5002.5 2204.83  5004.7 2207.65  5010.0 2207.65  5019.7 2223.53  5025.0 2241.20
  5030.2 2243.92  5065.5 2251.37  5071.4 2254.32  5081.7 2257.77  5100.7 2262.59
  5105.9 2261.80  5112.7 2263.62  5141.1 2267.99  5146.3 2267.54  5171.0 2270.50
#Mann=3,-1,0
  4879.1    0.16       0  4998.5    0.07       0  5002.5    0.16       0
Bank Sta=4998.5,5002.5
Exp/Cntr=0.3,0.1

Type RM Length L Ch R = 1,3186,17,17,17
BEGIN DESCRIPTION:
elmc562
END DESCRIPTION:
XS GIS Cut Line= 3
      1511779.61      6771968.24      1511861.02      6771896.60
      1511893.57      6771722.97
#Sta/Elev= 30
  4890.3 2263.70  4894.5 2261.20  4901.2 2260.32  4908.8 2257.70  4937.2 2250.01
  4943.9 2247.45  4950.8 2243.55  4964.8 2232.03  4972.3 2220.74  4979.0 2214.08
  4984.6 2204.34  4984.8 2203.84  4988.3 2203.84  4988.6 2204.34  4993.2 2204.69
  4998.1 2214.24  5007.5 2221.23  5017.7 2225.82  5045.3 2246.22  5050.4 2246.53
  5058.4 2249.28  5068.5 2251.50  5088.9 2254.18  5109.2 2258.39  5139.8 2261.68
  5149.9 2263.30  5155.5 2264.85  5160.6 2263.27  5170.3 2265.07  5175.4 2266.83
#Mann=3,-1,0
  4890.3    0.16       0  4984.6    0.07       0  4988.6    0.16       0
Bank Sta=4984.6,4988.6
Exp/Cntr=0.3,0.1

Type RM Length L Ch R = 1,3169,22,22,22
BEGIN DESCRIPTION:
elmc564
END DESCRIPTION:
XS GIS Cut Line= 3
      1511794.84      6771967.12      1511875.12      6771905.28
      1511972.76      6771746.89
#Sta/Elev= 30
  4901.4 2258.83  4928.8 2251.83  4943.4 2246.65  4957.9 2237.30  4972.4 2217.33
  4978.7 2211.42  4984.9 2200.81  4985.1 2200.31  4988.9 2200.81  4999.5 2207.97
  5002.7 2207.97  5008.7 2218.87  5023.0 2229.92  5045.4 2237.37  5051.3 2237.30
  5066.7 2245.67  5072.6 2242.40  5088.0 2242.95  5093.8 2238.43  5103.4 2239.95
  5109.2 2243.48  5124.6 2247.33  5130.5 2252.20  5140.0 2253.58  5145.9 2258.74
  5161.3 2259.34  5167.2 2264.36  5182.6 2264.33  5186.2 2268.52  5188.8 2268.52
#Mann=3,-1,0
  4901.4    0.16       0  4984.9    0.07       0  4988.9    0.16       0
Bank Sta=4984.9,4988.9
Exp/Cntr=0.3,0.1

Type RM Length L Ch R = 1,3147,24,24,24
BEGIN DESCRIPTION:
elmc563
END DESCRIPTION:
XS GIS Cut Line= 3
      1511799.19      6771973.63      1511885.97      6771926.98
      1511980.59      6771783.97
#Sta/Elev= 30
  4896.3 2258.78  4903.1 2256.17  4919.3 2252.44  4941.2 2244.13  4957.5 2228.07
  4963.2 2223.91  4971.0 2210.88  4983.1 2200.08  4983.3 2199.58  4987.1 2200.08
  4991.4 2202.33  4997.2 2202.33  5006.9 2213.29  5015.9 2219.69  5021.9 2226.10
  5029.6 2230.95  5052.0 2234.05  5058.0 2230.69  5065.5 2235.94  5073.1 2238.30
  5079.1 2234.95  5088.1 2236.27  5109.2 2245.14  5115.2 2249.61  5124.2 2252.49
  5130.2 2257.04  5145.3 2262.26  5151.3 2266.20  5160.3 2267.09  5166.3 2268.90
#Mann=3,-1,0
  4896.3    0.16       0  4983.1    0.07       0  4987.1    0.16       0
Bank Sta=4983.1,4987.1
Exp/Cntr=0.3,0.1

Type RM Length L Ch R = 1,3123,23,23,23
BEGIN DESCRIPTION:
elmc553
END DESCRIPTION:
XS GIS Cut Line= 3
      1511807.83      6772015.97      1511912.02      6771934.58
      1512000.63      6771813.93
#Sta/Elev= 30
  4875.7 2263.28  4879.5 2259.87  4922.9 2246.57  4929.2 2242.12  4935.6 2242.10
  4943.7 2231.14  4950.0 2227.25  4964.5 2215.47  4972.6 2205.95  4979.0 2200.46
  4984.3 2199.28  4984.6 2198.78  4988.3 2199.28  4993.4 2204.24  4999.8 2207.71
  5028.5 2219.14  5036.5 2224.99  5042.7 2225.55  5051.1 2228.75  5057.3 2234.92
  5072.0 2236.74  5078.2 2241.35  5086.6 2242.18  5092.8 2247.00  5101.3 2248.00
  5107.5 2253.63  5122.1 2256.61  5128.3 2263.24  5143.0 2266.52  5157.6 2268.12
#Mann=3,-1,0
  4875.7    0.16       0  4984.3    0.07       0  4988.3    0.16       0
Bank Sta=4984.3,4988.3
Exp/Cntr=0.3,0.1

Type RM Length L Ch R = 1,3100,24,24,24
BEGIN DESCRIPTION:
elmc552
END DESCRIPTION:
XS GIS Cut Line= 3
      1511828.45      6772022.48      1511918.53      6771959.53
      1512012.95      6771857.51
#Sta/Elev= 30
  4884.8 2256.70  4900.1 2250.27  4921.0 2243.63  4935.9 2229.78  4950.7 2220.58
  4956.8 2217.65  4965.5 2210.86  4971.6 2205.69  4976.2 2197.45  4976.4 2196.95
  4980.2 2197.45  4986.5 2198.00  4991.7 2203.21  4994.7 2203.21  5007.6 2208.62
  5014.4 2210.34  5021.8 2214.10  5028.6 2215.43  5035.9 2221.37  5042.7 2225.27
  5050.1 2231.56  5064.3 2241.62  5071.1 2244.13  5078.5 2245.60  5085.3 2248.47
  5092.2 2249.27  5106.3 2256.02  5113.6 2261.53  5127.8 2264.84  5133.7 2265.07
#Mann=3,-1,0
  4884.8    0.16       0  4976.2    0.07       0  4980.2    0.16       0
Bank Sta=4976.2,4980.2
Exp/Cntr=0.3,0.1

Type RM Length L Ch R = 1,3076,32,32,32
BEGIN DESCRIPTION:
elmc548
END DESCRIPTION:
XS GIS Cut Line= 3
      1511829.57      6772039.82      1511942.40      6771970.38
      1512030.42      6771883.44
#Sta/Elev= 30
  4871.4 2261.36  4877.8 2258.59  4889.9 2252.77  4899.4 2249.72  4905.3 2247.13
  4913.0 2242.58  4926.6 2233.87  4936.1 2228.83  4948.2 2220.47  4957.4 2215.09
  4963.3 2209.73  4976.7 2196.53  4976.9 2196.03  4980.4 2196.03  4980.7 2196.53
  4984.6 2199.28  4994.1 2202.54  5000.0 2204.07  5002.5 2206.98  5009.1 2206.98
  5035.7 2217.09  5063.9 2239.83  5078.1 2246.41  5085.2 2248.36  5092.2 2251.91
  5099.3 2254.50  5106.4 2258.05  5113.5 2259.31  5120.5 2261.57  5127.6 2262.64
#Mann=3,-1,0
  4871.4    0.16       0  4976.7    0.07       0  4980.7    0.16       0
Bank Sta=4976.7,4980.7
Exp/Cntr=0.3,0.1

Type RM Length L Ch R = 1,3044,36,36,36
BEGIN DESCRIPTION:
elmc549
END DESCRIPTION:
XS GIS Cut Line= 3
      1511850.15      6772069.13      1511960.84      6771996.43
      1512045.47      6771896.61
#Sta/Elev= 30
  4865.8 2259.28  4871.4 2259.28  4898.3 2247.81  4907.5 2247.31  4913.4 2243.10
  4928.5 2239.54  4934.5 2232.12  4943.4 2229.43  4949.6 2225.08  4955.6 2217.02
  4964.7 2208.55  4970.7 2200.60  4979.3 2195.29  4983.8 2194.66  4984.0 2194.16
  4987.8 2194.66  4991.7 2199.39  5000.5 2200.59  5007.6 2205.95  5014.1 2207.12
  5021.8 2211.26  5042.7 2223.43  5049.2 2229.47  5063.5 2239.34  5092.1 2254.19
  5099.8 2253.88  5114.1 2258.03  5120.7 2257.46  5124.9 2260.36  5129.1 2260.36
#Mann=3,-1,0
  4865.8    0.16       0  4983.8    0.07       0  4987.8    0.16       0
Bank Sta=4983.8,4987.8
Exp/Cntr=0.3,0.1

Type RM Length L Ch R = 1,3008,18,18,18
BEGIN DESCRIPTION:
elmc547
END DESCRIPTION:
XS GIS Cut Line= 3
      1511868.58      6772086.50      1511985.80      6772023.55
      1512062.85      6771907.44
#Sta/Elev= 30
  4863.4 2259.89  4867.9 2257.07  4889.8 2252.77  4895.5 2250.54  4904.7 2249.28
  4927.4 2241.47  4949.9 2226.50  4961.5 2212.02  4971.8 2203.19  4977.5 2197.09
  4982.2 2193.92  4982.4 2193.42  4986.2 2193.92  4996.4 2194.48  5000.6 2196.68
  5015.1 2200.17  5021.6 2204.06  5036.7 2217.75  5042.7 2220.73  5057.7 2232.24
  5072.8 2241.85  5078.8 2243.81  5093.8 2252.75  5099.8 2251.90  5108.8 2253.09
  5114.8 2250.97  5123.1 2252.99  5129.9 2256.03  5133.2 2253.90  5135.8 2253.90
#Mann=3,-1,0
  4863.4    0.16       0  4982.2    0.07       0  4986.2    0.16       0
Bank Sta=4982.2,4986.2
Exp/Cntr=0.3,0.1

Type RM Length L Ch R = 1,2990,22,22,22
BEGIN DESCRIPTION:
elmc550
END DESCRIPTION:
XS GIS Cut Line= 3
      1511891.40      6772093.00      1511998.82      6772034.40
      1512109.47      6771912.90
#Sta/Elev= 30
  4875.6 2253.74  4880.5 2253.74  4896.6 2251.38  4918.5 2244.06  4940.3 2231.18
  4956.4 2218.23  4962.1 2211.04  4978.3 2197.30  4982.0 2193.32  4982.2 2192.82
  4986.0 2193.32  5014.0 2197.72  5020.7 2203.89  5028.2 2206.39  5034.9 2212.83
  5042.4 2218.82  5049.1 2221.15  5056.5 2226.32  5063.3 2227.56  5070.7 2233.13
  5077.5 2234.77  5084.9 2241.87  5091.7 2242.49  5099.1 2245.33  5105.9 2242.61
  5113.3 2244.37  5120.1 2243.60  5141.7 2250.72  5148.4 2255.77  5162.3 2258.04
#Mann=3,-1,0
  4875.6    0.16       0  4982.0    0.07       0  4986.0    0.16       0
Bank Sta=4982,4986
Exp/Cntr=0.3,0.1

Type RM Length L Ch R = 1,2968,13,13,13
BEGIN DESCRIPTION:
elmc551
END DESCRIPTION:
XS GIS Cut Line= 3
      1511894.69      6772100.58      1512020.52      6772046.34
      1512120.70      6771934.32
#Sta/Elev= 30
  4868.1 2252.98  4879.3 2250.19  4886.0 2246.93  4891.4 2248.85  4909.5 2241.95
  4915.0 2242.28  4938.5 2229.57  4955.6 2216.62  4967.5 2202.65  4983.5 2193.30
  4983.8 2192.80  4987.5 2193.30  4991.0 2194.19  4999.1 2201.07  5007.4 2203.71
  5014.5 2208.78  5021.2 2209.57  5028.7 2214.61  5049.6 2221.13  5070.5 2225.35
  5084.7 2231.56  5092.2 2236.44  5106.4 2240.37  5113.1 2243.77  5120.6 2245.15
  5127.3 2248.92  5134.8 2251.19  5141.6 2255.74  5149.1 2258.22  5155.4 2261.83
#Mann=3,-1,0
  4868.1    0.16       0  4983.5    0.07       0  4987.5    0.16       0
Bank Sta=4983.5,4987.5
Exp/Cntr=0.3,0.1

Type RM Length L Ch R = 1,2955,39,39,39
BEGIN DESCRIPTION:
elmc398
END DESCRIPTION:
XS GIS Cut Line= 3
      1511904.44      6772103.84      1512025.39      6772057.84
      1512105.00      6771988.00
#Sta/Elev= 30
  4870.6 2247.26  4874.8 2250.19  4899.5 2239.38  4904.9 2241.95  4924.3 2233.97
  4929.6 2232.97  4935.4 2227.84  4954.4 2218.62  4959.7 2209.34  4967.5 2200.13
  4978.2 2193.48  4982.5 2192.36  4982.8 2191.86  4986.5 2192.36  4989.9 2195.14
  4997.1 2197.61  5003.1 2197.61  5006.7 2201.80  5013.4 2205.83  5035.2 2214.51
  5041.9 2218.61  5056.1 2222.28  5063.7 2227.30  5070.3 2228.93  5077.9 2234.39
  5084.6 2235.98  5092.1 2240.94  5098.8 2242.21  5102.6 2245.90  5105.9 2245.90
#Mann=3,-1,0
  4870.6    0.16       0  4982.5    0.07       0  4986.5    0.16       0
Bank Sta=4982.5,4986.5
Exp/Cntr=0.3,0.1

Type RM Length L Ch R = 1,2916,46,46,46
BEGIN DESCRIPTION:
elmc546
END DESCRIPTION:
XS GIS Cut Line= 3
      1511896.86      6772157.00      1512055.24      6772085.40
      1512164.46      6772001.89
#Sta/Elev= 30
  4832.3 2251.10  4838.9 2245.83  4852.2 2237.50  4867.5 2231.58  4874.2 2228.12
  4885.1 2226.67  4890.6 2228.26  4913.7 2222.54  4919.2 2224.58  4936.8 2218.77
  4942.3 2219.27  4951.0 2214.23  4965.4 2203.90  4972.9 2196.78  4983.0 2191.00
  4986.5 2190.37  4986.8 2189.87  4990.5 2190.37  5003.2 2205.67  5006.1 2205.67
  5011.1 2207.76  5025.6 2211.03  5040.1 2215.80  5054.7 2221.85  5068.8 2229.61
  5096.3 2248.50  5104.5 2252.60  5110.8 2254.96  5139.9 2258.58  5143.6 2260.02
#Mann=3,-1,0
  4832.3    0.16       0  4986.5    0.07       0  4990.5    0.16       0
Bank Sta=4986.5,4990.5
Exp/Cntr=0.3,0.1

Type RM Length L Ch R = 1,2870,27,27,27
BEGIN DESCRIPTION:
elmc545
END DESCRIPTION:
XS GIS Cut Line= 3
      1511921.81      6772204.75      1512048.73      6772141.83
      1512184.36      6772030.07
#Sta/Elev= 30
  4844.2 2250.33  4850.7 2249.40  4867.6 2240.28  4873.2 2239.63  4881.2 2235.14
  4912.4 2222.53  4934.8 2216.06  4940.4 2215.90  4948.2 2213.65  4957.3 2207.03
  4962.8 2205.95  4970.5 2199.20  4979.7 2193.64  4991.6 2189.23  4991.9 2188.73
  4995.4 2188.73  4995.6 2189.23  5000.1 2189.36  5014.4 2198.70  5020.9 2204.55
  5028.8 2205.40  5035.3 2208.66  5063.9 2215.84  5084.8 2225.61  5092.6 2230.40
  5113.5 2245.42  5127.8 2252.30  5142.1 2255.09  5149.5 2255.36  5161.6 2257.00
#Mann=3,-1,0
  4844.2    0.16       0  4991.6    0.07       0  4995.6    0.16       0
Bank Sta=4991.6,4995.6
Exp/Cntr=0.3,0.1

Type RM Length L Ch R = 1,2843,44,44,44
BEGIN DESCRIPTION:
elmc544
END DESCRIPTION:
XS GIS Cut Line= 3
      1511931.55      6772243.82      1512074.78      6772154.85
      1512188.70      6772043.09
#Sta/Elev= 30
  4832.9 2257.86  4838.7 2252.77  4848.1 2251.40  4854.0 2246.69  4860.5 2246.34
  4869.4 2243.14  4875.3 2238.41  4890.6 2229.29  4896.5 2226.67  4911.9 2222.13
  4927.2 2216.02  4969.7 2207.61  4978.2 2206.65  4985.1 2202.26  4991.0 2196.80
  4996.7 2188.91  4997.0 2188.41  5000.7 2188.91  5006.5 2189.00  5013.6 2192.23
  5020.6 2197.46  5034.8 2205.98  5063.1 2215.19  5091.4 2226.84  5098.5 2231.97
  5112.6 2239.02  5119.6 2244.88  5133.8 2251.98  5155.0 2255.00  5161.1 2255.00
#Mann=3,-1,0
  4832.9    0.16       0  4996.7    0.07       0  5000.7    0.16       0
Bank Sta=4996.7,5000.7
Exp/Cntr=0.3,0.1

Type RM Length L Ch R = 1,2799,39,39,39
BEGIN DESCRIPTION:
elmc543
END DESCRIPTION:
XS GIS Cut Line= 3
      1511952.15      6772257.94      1512104.07      6772188.48
      1512215.86      6772064.75
#Sta/Elev= 30
  4836.5 2254.34  4840.8 2254.34  4846.8 2249.73  4869.8 2240.68  4883.6 2232.03
  4905.6 2221.47  4921.3 2216.41  4927.6 2213.31  4938.6 2210.31  4944.3 2207.55
  4949.8 2207.70  4960.6 2205.87  4990.4 2199.29  4995.9 2193.42  4999.3 2187.74
  4999.6 2187.24  5003.3 2187.74  5011.7 2188.23  5025.9 2195.52  5040.1 2201.24
  5054.3 2208.40  5075.2 2221.73  5082.6 2225.25  5103.6 2232.81  5125.2 2244.54
  5139.0 2250.51  5146.2 2252.58  5152.9 2252.59  5160.4 2254.62  5170.3 2254.65
#Mann=3,-1,0
  4836.5    0.16       0  4999.3    0.07       0  5003.3    0.16       0
Bank Sta=4999.3,5003.3
Exp/Cntr=0.3,0.1

Type RM Length L Ch R = 1,2760,46,46,46
BEGIN DESCRIPTION:
elmc542
END DESCRIPTION:
XS GIS Cut Line= 3
      1511968.48      6772294.80      1512110.58      6772226.46
      1512263.60      6772127.70
#Sta/Elev= 30
  4846.4 2261.18  4849.3 2259.24  4864.7 2254.49  4872.0 2251.44  4886.9 2242.89
  4894.6 2237.65  4939.8 2214.58  4945.4 2212.97  4962.5 2205.08  4985.1 2199.94
  4990.7 2199.74  4997.9 2195.65  5003.8 2190.86  5012.9 2190.12  5019.2 2185.45
  5019.5 2184.95  5023.2 2185.45  5034.0 2188.83  5056.9 2202.21  5070.3 2208.94
  5085.5 2212.81  5106.6 2216.92  5121.8 2221.21  5152.1 2238.99  5158.0 2241.55
  5164.1 2245.76  5173.2 2249.42  5179.2 2249.60  5184.0 2253.33  5186.2 2253.33
#Mann=3,-1,0
  4846.4    0.16       0  5019.2    0.07       0  5023.2    0.16       0
Bank Sta=5019.2,5023.2
Exp/Cntr=0.3,0.1

Type RM Length L Ch R = 1,2714,51,51,51
BEGIN DESCRIPTION:
elmc541
END DESCRIPTION:
XS GIS Cut Line= 3
      1512017.28      6772336.04      1512134.45      6772264.44
      1512275.55      6772170.01
#Sta/Elev= 30
  4864.3 2257.52  4874.7 2250.25  4884.3 2246.22  4920.2 2221.82  4926.9 2215.97
  4963.6 2200.67  4969.5 2200.18  4978.8 2197.15  4984.9 2191.79  4990.8 2191.21
  4999.0 2185.24  5004.3 2184.95  5004.5 2184.45  5008.3 2184.95  5014.3 2187.27
  5021.3 2192.39  5036.3 2197.99  5042.3 2199.54  5057.3 2199.82  5063.3 2202.16
  5072.3 2203.71  5078.3 2207.79  5093.3 2212.60  5099.3 2216.29  5122.6 2225.15
  5135.4 2231.79  5150.4 2241.74  5158.7 2245.00  5168.7 2250.95  5171.4 2250.95
#Mann=3,-1,0
  4864.3    0.16       0  5004.3    0.07       0  5008.3    0.16       0
Bank Sta=5004.3,5008.3
Exp/Cntr=0.3,0.1

Type RM Length L Ch R = 1,2663,49,49,49
BEGIN DESCRIPTION:
elmc540
END DESCRIPTION:
XS GIS Cut Line= 3
      1512044.41      6772375.11      1512164.84      6772304.59
      1512299.15      6772202.77
#Sta/Elev= 30
  4855.5 2255.39  4867.8 2252.30  4876.5 2248.82  4903.8 2225.35  4913.7 2220.33
  4925.7 2210.84  4941.0 2203.71  4956.6 2194.51  4962.4 2192.57  4972.1 2186.85
  4978.1 2181.22  4981.9 2181.18  4982.2 2180.68  4985.9 2181.18  4995.1 2183.06
  4999.6 2185.34  5007.8 2192.43  5057.8 2196.90  5078.6 2202.26  5084.9 2205.98
  5093.2 2208.75  5099.5 2212.95  5107.7 2215.44  5114.0 2219.77  5128.6 2225.83
  5134.8 2231.08  5143.1 2236.06  5149.4 2242.16  5157.7 2245.19  5163.6 2248.73
#Mann=3,-1,0
  4855.5    0.16       0  4981.9    0.07       0  4985.9    0.16       0
Bank Sta=4981.9,4985.9
Exp/Cntr=0.3,0.1

Type RM Length L Ch R = 1,2614,35,35,35
BEGIN DESCRIPTION:
elmc538
END DESCRIPTION:
XS GIS Cut Line= 3
      1512058.46      6772407.69      1512199.56      6772339.31
      1512326.51      6772232.97
#Sta/Elev= 30
  4838.7 2253.80  4867.5 2248.53  4873.1 2245.03  4879.3 2239.22  4895.6 2227.66
  4901.5 2221.15  4912.6 2215.26  4918.2 2209.40  4934.9 2200.93  4940.8 2195.45
  4957.1 2186.30  4963.4 2179.13  4977.3 2175.14  4977.6 2174.64  4981.3 2175.14
  4986.0 2178.84  4991.3 2184.16  5000.7 2183.16  5007.2 2187.11  5015.0 2183.08
  5021.5 2187.93  5035.8 2193.13  5050.1 2195.33  5078.8 2202.08  5085.3 2204.89
  5113.9 2221.50  5120.4 2224.17  5142.5 2237.44  5149.0 2240.09  5161.1 2243.06
#Mann=3,-1,0
  4838.7    0.16       0  4977.3    0.07       0  4981.3    0.16       0
Bank Sta=4977.3,4981.3
Exp/Cntr=0.3,0.1

Type RM Length L Ch R = 1,2579,36,36,36
BEGIN DESCRIPTION:
elmc539
END DESCRIPTION:
XS GIS Cut Line= 3
      1512086.73      6772415.26      1512232.11      6772359.92
      1512347.16      6772245.96
#Sta/Elev= 30
  4849.1 2244.95  4854.0 2238.95  4859.4 2240.71  4878.8 2226.94  4884.1 2226.08
  4890.1 2219.37  4908.9 2207.10  4914.2 2205.94  4922.2 2200.58  4932.9 2195.91
  4944.3 2189.15  4963.7 2181.85  4969.1 2176.17  4991.9 2171.64  4992.1 2171.14
  4995.9 2171.64  4999.2 2175.75  5003.5 2178.25  5009.6 2178.25  5015.1 2184.76
  5022.2 2190.38  5057.6 2195.66  5071.7 2200.89  5128.3 2229.68  5135.4 2229.70
  5142.4 2237.18  5149.5 2236.19  5156.6 2229.71  5161.6 2232.73  5166.6 2232.73
#Mann=3,-1,0
  4849.1    0.16       0  4991.9    0.07       0  4995.9    0.16       0
Bank Sta=4991.9,4995.9
Exp/Cntr=0.3,0.1

Type RM Length L Ch R = 1,2543,49,49,49
BEGIN DESCRIPTION:
elmc536
END DESCRIPTION:
XS GIS Cut Line= 3
      1512061.76      6772435.88      1512254.90      6772388.14
      1512420.45      6772250.72
#Sta/Elev= 30
  4806.1 2249.36  4810.3 2249.36  4816.3 2245.54  4821.5 2248.17  4850.6 2229.65
  4857.8 2223.28  4862.9 2225.36  4899.2 2202.29  4904.4 2202.26  4912.4 2197.39
  4940.6 2186.71  4953.6 2184.12  4992.9 2171.65  4993.1 2171.15  4996.9 2171.65
  5002.5 2177.37  5008.4 2177.37  5012.4 2184.06  5026.7 2192.76  5069.7 2198.17
  5097.0 2209.16  5111.3 2213.19  5125.7 2214.69  5133.5 2213.83  5140.0 2216.07
  5147.8 2215.42  5168.6 2220.95  5203.8 2241.67  5211.6 2241.91  5220.2 2247.12
#Mann=3,-1,0
  4806.1    0.16       0  4992.9    0.07       0  4996.9    0.16       0
Bank Sta=4992.9,4996.9
Exp/Cntr=0.3,0.1

Type RM Length L Ch R = 1,2494,30,30,30
BEGIN DESCRIPTION:
elmc537
END DESCRIPTION:
XS GIS Cut Line= 3
      1512091.02      6772502.08      1512258.15      6772436.96
      1512475.15      6772333.89
#Sta/Elev= 30
  4819.6 2244.88  4824.4 2244.88  4830.4 2240.15  4847.7 2223.53  4877.5 2206.00
  4909.7 2198.69  4937.8 2194.53  4956.4 2192.16  4963.4 2189.41  4994.6 2173.06
  4999.0 2173.06  5002.6 2169.01  5002.9 2168.51  5006.6 2169.01  5010.1 2169.86
  5027.3 2182.13  5032.9 2184.19  5039.8 2190.36  5078.3 2196.21  5101.0 2196.70
  5123.8 2199.41  5129.3 2201.88  5139.4 2202.80  5161.5 2209.21  5169.2 2213.84
  5174.8 2214.41  5191.9 2221.00  5205.8 2223.11  5220.2 2223.33  5239.2 2226.88
#Mann=5,-1,0
  4819.6    0.16       0  4830.4    0.07       0  4937.8    0.16       0
  5002.6    0.07       0  5006.6    0.16       0
Bank Sta=5002.6,5006.6
Exp/Cntr=0.3,0.1

Type RM Length L Ch R = 1,2464,87,87,87
BEGIN DESCRIPTION:
elmc535
END DESCRIPTION:
XS GIS Cut Line= 3
      1512145.33      6772548.71      1512280.94      6772458.67
      1512461.03      6772381.02
#Sta/Elev= 30
  4840.8 2239.16  4843.6 2239.16  4854.8 2227.20  4863.8 2223.26  4869.8 2218.39
  4890.8 2206.33  4906.0 2200.64  4957.0 2189.47  4963.0 2184.98  4972.1 2183.25
  4984.4 2174.64  4997.1 2168.38  4997.3 2167.88  5001.1 2168.38  5003.0 2172.57
  5008.5 2172.57  5029.8 2186.35  5044.6 2190.16  5068.2 2188.82  5073.6 2192.20
  5106.0 2195.29  5120.6 2198.71  5138.7 2209.59  5144.2 2215.46  5149.6 2215.79
  5167.7 2227.26  5173.1 2225.71  5191.2 2235.47  5196.6 2233.57  5199.7 2237.55
#Mann=4,-1,0
  4840.8    0.07       0  4906.0    0.16       0  4997.1    0.07       0
  5001.1    0.16       0
Bank Sta=4997.1,5001.1
Exp/Cntr=0.3,0.1

Type RM Length L Ch R = 1,2377,62,62,62
BEGIN DESCRIPTION:
elmc534
END DESCRIPTION:
XS GIS Cut Line= 3
      1512208.23      6772605.16      1512336.28      6772524.85
      1512458.89      6772408.76
#Sta/Elev= 30
  4845.2 2233.06  4848.3 2227.65  4863.6 2220.18  4869.5 2219.00  4884.8 2209.80
  4906.0 2203.80  4921.3 2194.33  4943.5 2185.57  4979.1 2173.69  4985.0 2169.82
  4996.3 2168.45  5000.3 2165.61  5005.5 2165.00  5005.8 2164.50  5009.5 2165.00
  5035.8 2175.37  5049.7 2184.74  5063.8 2188.24  5071.0 2187.89  5085.2 2193.24
  5092.1 2197.84  5113.5 2206.44  5120.4 2211.54  5127.7 2213.24  5134.6 2218.84
  5141.8 2220.31  5148.7 2225.57  5156.0 2225.95  5162.1 2230.73  5165.2 2230.73
#Mann=4,-1,0
  4845.2    0.07       0  4943.5    0.16       0  5005.5    0.07       0
  5009.5    0.16       0
Bank Sta=5005.5,5009.5
Exp/Cntr=0.3,0.1

Type RM Length L Ch R = 1,2315,75,75,75
BEGIN DESCRIPTION:
elmc533
END DESCRIPTION:
XS GIS Cut Line= 3
      1512317.83      6772632.28      1512382.94      6772566.09
      1512458.88      6772446.75
#Sta/Elev= 30
  4907.7 2218.02  4922.9 2210.75  4937.0 2202.38  4944.0 2200.06  4958.2 2188.91
  4965.3 2187.50  4972.3 2181.86  4979.5 2179.48  4986.5 2175.74  4998.5 2170.91
  5009.0 2168.98  5013.0 2166.21  5014.9 2164.89  5020.0 2163.78  5020.2 2163.28
  5024.0 2163.78  5036.0 2172.06  5051.3 2178.03  5057.5 2183.01  5066.5 2185.31
  5072.5 2184.46  5081.3 2185.38  5087.7 2187.92  5093.6 2188.28  5102.9 2193.00
  5108.9 2193.30  5124.1 2203.31  5130.0 2203.62  5138.3 2209.11  5142.0 2209.11
#Mann=4,-1,0
  4907.7    0.07       0  5013.0    0.16       0  5020.0    0.07       0
  5024.0    0.16       0
Bank Sta=5020,5024
Exp/Cntr=0.3,0.1

Type RM Length L Ch R = 1,2240,65,65,65
BEGIN DESCRIPTION:
elmc532
END DESCRIPTION:
XS GIS Cut Line= 3
      1512331.91      6772658.33      1512432.85      6772621.43
      1512578.26      6772530.27
#Sta/Elev= 30
  4889.6 2218.22  4893.9 2218.22  4901.7 2214.75  4907.0 2215.26  4924.8 2206.04
  4937.5 2196.75  4955.8 2189.45  4962.7 2184.59  4978.1 2177.01  4987.9 2170.82
  4993.3 2166.21  4995.6 2162.13  5007.2 2161.81  5007.5 2161.31  5011.2 2161.81
  5015.1 2164.89  5036.3 2171.31  5058.6 2180.26  5067.0 2182.17  5072.9 2181.06
  5088.2 2184.87  5094.1 2183.69  5103.5 2185.58  5109.4 2184.48  5124.7 2188.68
  5130.6 2188.39  5145.9 2189.74  5153.0 2190.92  5161.3 2193.81  5168.7 2194.03
#Mann=4,-1,0
  4889.6    0.07       0  4955.8    0.16       0  5007.2    0.07       0
  5011.2    0.16       0
Bank Sta=5007.2,5011.2
Exp/Cntr=0.3,0.1

Type RM Length L Ch R = 1,2175,56,56,56
BEGIN DESCRIPTION:
elmc531
END DESCRIPTION:
XS GIS Cut Line= 3
      1512337.34      6772704.98      1512451.29      6772680.02
      1512583.70      6772618.16
#Sta/Elev= 30
  4879.5 2216.28  4885.5 2211.10  4890.6 2211.55  4897.6 2206.40  4918.1 2196.31
  4928.3 2190.76  4934.5 2186.38  4936.0 2186.81  4939.6 2187.84  4948.8 2184.76
  4959.0 2179.87  4978.3 2168.05  4983.4 2168.82  4989.7 2164.26  4993.5 2159.37
  4993.7 2158.87  4997.2 2158.87  4997.5 2159.37  5009.3 2160.59  5014.8 2159.66
  5022.3 2166.48  5032.1 2172.79  5037.6 2172.62  5055.0 2178.56  5060.5 2176.74
  5083.3 2183.88  5088.8 2184.94  5106.2 2186.45  5134.5 2191.24  5142.3 2192.04
#Mann=4,-1,0
  4879.5    0.07       0  4936.0    0.16       0  4993.5    0.07       0
  4997.5    0.16       0
Bank Sta=4993.5,4997.5
Exp/Cntr=0.3,0.1

Type RM Length L Ch R = 1,2119,66,66,66
BEGIN DESCRIPTION:
elmc530
END DESCRIPTION:
XS GIS Cut Line= 3
      1512325.38      6772792.89      1512451.29      6772737.53
      1512649.86      6772643.13
#Sta/Elev= 30
  4854.6 2217.98  4857.1 2217.98  4887.0 2197.73  4903.7 2188.65  4909.1 2188.35
  4925.7 2184.03  4932.5 2183.78  4941.6 2181.46  4955.8 2179.53  4963.4 2177.62
  4973.7 2173.19  4979.2 2169.23  4985.3 2162.78  4989.4 2156.64  4989.7 2156.14
  4993.2 2156.14  4993.4 2156.64  4997.0 2156.64  5007.8 2163.41  5018.4 2166.52
  5023.9 2170.47  5047.7 2179.80  5053.2 2177.98  5062.7 2180.94  5098.6 2183.40
  5107.0 2184.69  5173.4 2191.36  5189.5 2194.64  5206.5 2200.24  5212.0 2200.24
#Mann=4,-1,0
  4854.6    0.07       0  4925.7    0.16       0  4989.4    0.07       0
  4993.4    0.16       0
Bank Sta=4989.4,4993.4
Exp/Cntr=0.3,0.1

Type RM Length L Ch R = 1,2053,56,56,56
BEGIN DESCRIPTION:
elmc529
END DESCRIPTION:
XS GIS Cut Line= 3
      1512347.12      6772844.95      1512493.61      6772787.44
      1512647.54      6772732.54
#Sta/Elev= 30
  4837.2 2215.85  4841.4 2210.11  4846.8 2208.43  4881.8 2191.07  4888.6 2188.19
  4895.6 2183.14  4925.4 2178.73  4942.3 2175.15  4977.7 2158.04  4977.9 2157.54
  4981.7 2158.04  4985.3 2158.28  4992.6 2164.71  4998.0 2164.71  5004.6 2169.07
  5017.3 2175.16  5035.4 2180.90  5040.7 2180.12  5049.1 2181.22  5059.7 2183.13
  5066.2 2185.65  5081.0 2187.00  5097.0 2190.63  5102.3 2189.31  5112.8 2191.33
  5122.5 2194.84  5127.8 2192.27  5134.1 2195.00  5153.3 2198.28  5158.0 2196.62
#Mann=4,-1,0
  4837.2    0.07       0  4881.8    0.16       0  4977.7    0.07       0
  4981.7    0.16       0
Bank Sta=4977.7,4981.7
Exp/Cntr=0.3,0.1

Type RM Length L Ch R = 1,1997,60,60,60
BEGIN DESCRIPTION:
elmc397
END DESCRIPTION:
XS GIS Cut Line= 3
      1512355.02      6772937.99      1512511.11      6772840.18
      1512620.27      6772788.67
#Sta/Elev= 30
  4815.8 2222.47  4818.7 2222.47  4823.4 2219.44  4829.3 2218.75  4844.6 2212.79
  4852.5 2204.79  4860.0 2198.67  4881.2 2186.78  4896.5 2181.41  4902.4 2181.99
  4917.7 2177.73  4923.6 2178.20  4938.9 2175.80  4981.4 2156.06  4988.8 2154.83
  4989.0 2154.33  4992.8 2154.83  4996.7 2157.51  4999.3 2163.18  5013.3 2164.67
  5018.9 2169.86  5036.1 2172.79  5041.6 2179.05  5070.6 2192.96  5081.6 2196.77
  5087.2 2196.17  5092.8 2200.64  5109.9 2209.01  5115.5 2205.89  5120.7 2209.44
#Mann=4,-1,0
  4815.8    0.07       0  4852.5    0.16       0  4988.8    0.07       0
  4992.8    0.16       0
Bank Sta=4988.8,4992.8
Exp/Cntr=0.3,0.1

Type RM Length L Ch R = 1,1937,76,76,76
BEGIN DESCRIPTION:
elmc527
END DESCRIPTION:
XS GIS Cut Line= 3
      1512368.84      6772957.79      1512546.78      6772888.35
      1512649.84      6772826.52
#Sta/Elev= 30
  4806.5 2221.34  4813.1 2217.61  4819.1 2212.49  4824.1 2210.83  4843.6 2197.02
  4848.9 2196.26  4856.1 2190.39  4873.4 2181.04  4878.8 2179.04  4897.9 2175.76
  4941.9 2172.75  4957.6 2168.05  4963.4 2163.59  4991.9 2152.95  4992.1 2152.45
  4995.9 2152.95  5004.6 2153.59  5018.8 2166.74  5026.0 2176.14  5031.8 2175.65
  5041.5 2187.40  5047.4 2186.43  5053.7 2191.89  5062.9 2193.90  5068.7 2197.99
  5084.3 2202.81  5090.1 2207.68  5099.8 2209.25  5105.7 2214.27  5117.7 2215.03
#Mann=4,-1,0
  4806.5    0.07       0  4824.1    0.16       0  4991.9    0.07       0
  4995.9    0.16       0
Bank Sta=4991.9,4995.9
Exp/Cntr=0.3,0.1

Type RM Length L Ch R = 1,1861,61,61,61
BEGIN DESCRIPTION:
elmc528
END DESCRIPTION:
XS GIS Cut Line= 3
      1512384.05      6772989.26      1512554.38      6772962.14
      1512699.35      6772882.67
#Sta/Elev= 30
  4826.9 2213.46  4827.0 2213.46  4829.9 2213.46  4838.0 2208.88  4858.2 2195.60
  4865.0 2189.27  4870.1 2189.06  4878.5 2184.61  4898.7 2178.06  4932.2 2173.18
  4949.4 2164.31  4969.6 2151.20  4977.8 2149.02  4978.0 2148.52  4981.8 2149.02
  4989.4 2151.13  4997.2 2155.17  5017.8 2157.44  5023.5 2161.02  5045.7 2170.15
  5077.5 2171.98  5083.2 2173.52  5099.3 2173.60  5114.1 2175.99  5121.1 2175.37
  5126.8 2179.26  5142.9 2179.08  5148.6 2182.60  5159.0 2181.92  5164.7 2184.89
#Mann=4,-1,0
  4826.9    0.07       0  4827.0    0.16       0  4977.8    0.07       0
  4981.8    0.16       0
Bank Sta=4977.8,4981.8
Exp/Cntr=0.3,0.1

Type RM Length L Ch R = 1,1800,45,45,45
BEGIN DESCRIPTION:
elmc525
END DESCRIPTION:
XS GIS Cut Line= 3
      1512437.19      6773088.01      1512580.42      6773015.31
      1512811.85      6772925.96
#Sta/Elev= 30
  4838.3 2205.39  4845.4 2202.43  4851.0 2197.85  4867.7 2192.13  4895.5 2178.26
  4912.2 2174.81  4925.6 2174.09  4940.1 2169.91  4956.7 2169.38  4962.3 2166.67
  4979.0 2162.67  4984.6 2159.14  4998.7 2154.43  5007.3 2152.95  5012.6 2147.12
  5012.8 2146.62  5016.6 2147.12  5025.3 2147.70  5037.2 2156.32  5100.3 2159.21
  5141.0 2166.95  5146.4 2162.14  5153.9 2167.73  5164.6 2167.45  5171.0 2170.42
  5186.1 2173.17  5195.6 2178.55  5225.5 2182.95  5230.9 2182.53  5247.0 2185.73
#Mann=3,-1,0
  4838.3    0.16       0  5012.6    0.07       0  5016.6    0.16       0
Bank Sta=5012.6,5016.6
Exp/Cntr=0.3,0.1

Type RM Length L Ch R = 1,1755,55,55,55
BEGIN DESCRIPTION:
elmc526
END DESCRIPTION:
XS GIS Cut Line= 3
      1512469.76      6773107.53      1512617.31      6773044.60
      1512814.81      6772966.47
#Sta/Elev= 30
  4844.9 2198.75  4861.7 2188.41  4885.3 2179.23  4908.9 2176.14  4926.7 2177.04
  4932.5 2174.51  4948.4 2171.08  4956.1 2166.75  4961.6 2164.79  4970.2 2159.02
  4979.8 2154.24  4999.3 2146.04  4999.6 2145.54  5003.3 2146.04  5008.9 2146.04
  5024.3 2154.28  5033.3 2156.83  5038.7 2156.24  5045.8 2158.38  5087.3 2162.88
  5092.7 2166.38  5110.4 2165.48  5117.1 2168.24  5141.4 2175.29  5146.8 2174.69
  5153.4 2177.91  5185.6 2180.82  5200.9 2184.13  5207.1 2187.83  5217.7 2189.68
#Mann=3,-1,0
  4844.9    0.16       0  4999.3    0.07       0  5003.3    0.16       0
Bank Sta=4999.3,5003.3
Exp/Cntr=0.3,0.1

Type RM Length L Ch R = 1,1700,50,50,50
BEGIN DESCRIPTION:
elmc524
END DESCRIPTION:
XS GIS Cut Line= 3
      1512489.25      6773119.48      1512650.95      6773086.92
      1512810.19      6773004.59
#Sta/Elev= 30
  4836.7 2188.25  4842.6 2184.18  4868.8 2178.08  4873.9 2178.72  4893.6 2176.77
  4914.0 2171.77  4919.6 2169.18  4924.7 2168.91  4944.6 2160.75  4965.0 2154.30
  4970.5 2149.10  4975.6 2145.62  4983.4 2144.39  4983.6 2143.89  4987.4 2144.39
  4995.6 2148.34  5001.2 2153.28  5005.9 2153.28  5011.0 2154.31  5027.5 2154.19
  5055.3 2157.29  5071.8 2162.64  5077.4 2162.89  5085.0 2166.68  5094.0 2170.01
  5107.5 2173.55  5121.7 2174.79  5130.0 2176.62  5166.0 2180.70  5180.9 2183.53
#Mann=3,-1,0
  4836.7    0.16       0  4983.4    0.07       0  4987.4    0.16       0
Bank Sta=4983.4,4987.4
Exp/Cntr=0.3,0.1

Type RM Length L Ch R = 1,1650,63,63,63
BEGIN DESCRIPTION:
elmc523
END DESCRIPTION:
XS GIS Cut Line= 3
      1512475.17      6773175.90      1512655.29      6773136.83
      1512808.27      6773118.39
#Sta/Elev= 30
  4811.5 2183.07  4814.0 2183.07  4825.9 2180.38  4831.8 2179.76  4870.0 2178.30
  4875.1 2177.18  4893.2 2175.00  4903.4 2174.74  4914.7 2171.61  4919.2 2168.97
  4954.6 2166.64  4968.3 2164.27  4985.3 2155.65  4993.1 2150.12  4998.2 2150.12
  5005.6 2144.67  5013.7 2141.24  5013.9 2140.74  5017.4 2140.74  5017.7 2141.24
  5024.3 2144.73  5029.3 2149.11  5035.8 2153.67  5056.0 2156.33  5066.0 2156.94
  5096.2 2166.09  5106.3 2169.75  5111.4 2174.10  5145.7 2178.40  5149.9 2178.40
#Mann=4,-1,0
  4811.5    0.07       0  4914.7    0.16       0  5013.7    0.07       0
  5017.7    0.16       0
Bank Sta=5013.7,5017.7
Exp/Cntr=0.3,0.1

Type RM Length L Ch R = 1,1587,79,79,79
BEGIN DESCRIPTION:
elmc521
END DESCRIPTION:
XS GIS Cut Line= 3
      1512509.87      6773206.28      1512700.86      6773185.66
      1512870.64      6773173.77
#Sta/Elev= 30
  4812.2 2191.63  4817.4 2193.84  4827.4 2193.81  4837.5 2192.18  4847.7 2185.49
  4857.6 2183.55  4865.7 2181.17  4877.7 2177.65  4887.8 2173.70  4897.8 2169.16
  4917.9 2160.64  4928.0 2158.67  4934.5 2156.65  4939.5 2158.69  4958.2 2152.78
  4968.2 2150.67  4978.3 2147.39  4996.4 2140.08  4996.7 2139.58  5000.2 2139.58
  5000.4 2140.08  5003.9 2146.51  5008.9 2146.51  5018.5 2154.71  5043.0 2165.94
  5048.5 2171.18  5068.6 2172.72  5108.7 2177.39  5168.8 2182.79  5174.5 2184.32
#Mann=4,-1,0
  4812.2    0.07       0  4865.7    0.16       0  4996.4    0.07       0
  5000.4    0.16       0
Bank Sta=4996.4,5000.4
Exp/Cntr=0.3,0.1

Type RM Length L Ch R = 1,1508,52,52,52
BEGIN DESCRIPTION:
elmc522
END DESCRIPTION:
XS GIS Cut Line= 3
      1512522.89      6773244.26      1512654.20      6773252.94
      1512841.47      6773216.34
#Sta/Elev= 30
  4866.1 2197.22  4878.2 2196.30  4888.3 2193.26  4893.7 2190.78  4958.4 2161.60
  4978.5 2150.79  4988.5 2147.18  4995.6 2143.55  5000.6 2143.55  5008.7 2138.98
  5016.9 2138.09  5017.1 2137.59  5020.6 2137.59  5020.9 2138.09  5029.1 2138.24
  5039.3 2147.09  5046.9 2155.60  5052.0 2150.89  5059.6 2158.85  5069.8 2163.73
  5090.2 2166.28  5110.6 2169.73  5120.8 2170.20  5131.0 2172.70  5141.2 2173.96
  5150.0 2176.28  5155.1 2175.52  5161.5 2177.27  5181.9 2179.41  5188.5 2181.19
#Mann=4,-1,0
  4866.1    0.07       0  4893.7    0.16       0  5016.9    0.07       0
  5020.9    0.16       0
Bank Sta=5016.9,5020.9
Exp/Cntr=0.3,0.1

Type RM Length L Ch R = 1,1456,50,50,50
BEGIN DESCRIPTION:
elmc518
END DESCRIPTION:
XS GIS Cut Line= 3
      1512493.59      6773309.36      1512649.86      6773305.02
      1512831.62      6773255.55
#Sta/Elev= 30
  4838.1 2185.47  4859.5 2188.40  4869.5 2187.96  4877.6 2185.61  4919.5 2175.11
  4939.5 2167.30  4959.6 2156.74  4969.6 2150.08  4987.5 2136.05  4987.7 2135.55
  4991.5 2136.05  4994.4 2136.05  5003.5 2140.22  5010.1 2144.12  5020.5 2148.07
  5030.8 2149.47  5038.1 2153.71  5043.3 2153.50  5051.6 2156.70  5072.3 2160.45
  5077.9 2163.38  5083.1 2159.13  5093.0 2165.90  5112.5 2169.47  5117.6 2169.38
  5124.1 2171.55  5144.8 2175.41  5157.4 2179.15  5165.6 2180.66  5182.8 2181.51
#Mann=4,-1,0
  4838.1    0.07       0  4877.6    0.16       0  4987.5    0.07       0
  4991.5    0.16       0
Bank Sta=4987.5,4991.5
Exp/Cntr=0.3,0.1

Type RM Length L Ch R = 1,1406,51,51,51
BEGIN DESCRIPTION:
elmc520
END DESCRIPTION:
XS GIS Cut Line= 3
      1512452.36      6773428.73      1512663.97      6773352.76
      1512815.38      6773272.73
#Sta/Elev= 30
  4770.7 2184.41  4774.8 2184.41  4805.4 2172.16  4814.0 2170.01  4840.7 2169.83
  4890.4 2166.65  4954.1 2161.05  4962.3 2158.81  4986.0 2149.36  4993.1 2144.98
  4995.2 2141.17  4998.9 2141.17  5008.0 2135.41  5013.0 2134.71  5013.3 2134.21
  5017.0 2134.71  5030.6 2145.56  5037.1 2147.22  5042.7 2150.28  5059.1 2152.55
  5064.7 2157.28  5075.4 2158.65  5081.1 2161.68  5097.4 2162.87  5103.1 2165.09
  5119.4 2167.19  5132.4 2171.43  5147.1 2174.55  5163.5 2176.30  5166.8 2178.42
#Mann=4,-1,0
  4770.7    0.07       0  4840.7    0.16       0  5013.0    0.07       0
  5017.0    0.16       0
Bank Sta=5013,5017
Exp/Cntr=0.3,0.1

Type RM Length L Ch R = 1,1355,45,45,45
BEGIN DESCRIPTION:
elmc519
END DESCRIPTION:
XS GIS Cut Line= 3
      1512491.42      6773485.15      1512709.54      6773384.23
      1512838.67      6773275.72
#Sta/Elev= 30
  4765.7 2173.14  4795.9 2171.66  4802.7 2169.56  4813.3 2168.16  4853.1 2164.80
  4864.7 2163.81  4870.2 2162.43  4887.6 2161.78  4893.1 2162.52  4916.1 2161.26
  4979.0 2155.77  4984.8 2153.22  4990.3 2144.73  5006.0 2138.67  5011.8 2132.18
  5012.1 2131.68  5015.8 2132.18  5021.6 2133.60  5028.1 2138.86  5035.9 2141.01
  5042.4 2144.99  5050.2 2147.29  5071.0 2156.70  5099.6 2165.01  5134.8 2172.55
  5142.5 2172.21  5149.1 2174.21  5156.8 2174.68  5169.0 2177.18  5174.7 2177.18
#Mann=4,-1,0
  4765.7    0.07       0  4853.1    0.16       0  5011.8    0.07       0
  5015.8    0.16       0
Bank Sta=5011.8,5015.8
Exp/Cntr=0.3,0.1

Type RM Length L Ch R = 1,1310,54,54,54
BEGIN DESCRIPTION:
elmc517
END DESCRIPTION:
XS GIS Cut Line= 3
      1512585.80      6773512.29      1512737.75      6773416.78
      1512853.78      6773301.83
#Sta/Elev= 30
  4823.1 2162.61  4840.2 2161.01  4846.1 2161.76  4855.5 2159.63  4861.4 2160.08
  4876.7 2156.26  4882.6 2158.28  4919.1 2156.87  4934.4 2154.67  4976.9 2152.59
  4992.2 2147.84  4998.0 2140.95  5002.6 2140.95  5004.8 2132.70  5005.1 2132.20
  5008.8 2132.70  5021.0 2132.78  5028.0 2136.55  5035.1 2143.03  5056.3 2153.33
  5077.6 2156.88  5084.6 2159.10  5105.8 2160.62  5127.0 2164.59  5134.1 2164.23
  5141.2 2167.92  5148.3 2168.33  5155.3 2170.57  5162.4 2170.42  5165.9 2172.85
#Mann=3,-1,0
  4823.1    0.16       0  5004.8    0.07       0  5008.8    0.16       0
Bank Sta=5004.8,5008.8
Exp/Cntr=0.3,0.1

Type RM Length L Ch R = 1,1256,62,62,62
BEGIN DESCRIPTION:
elmc516
END DESCRIPTION:
XS GIS Cut Line= 3
      1512579.37      6773536.12      1512755.11      6773466.70
      1512907.07      6773424.37
#Sta/Elev= 30
  4810.9 2163.05  4815.5 2161.65  4822.2 2161.64  4838.5 2160.42  4869.6 2156.49
  4904.7 2155.10  4923.7 2152.22  4929.1 2152.70  4935.2 2147.27  4953.4 2144.22
  4958.8 2146.76  4967.5 2143.96  4977.8 2134.06  4983.2 2136.21  4987.0 2128.92
  4987.2 2128.42  4990.7 2128.42  4991.0 2128.92  4997.1 2136.05  5002.4 2136.05
  5009.3 2139.49  5014.5 2139.44  5020.5 2142.76  5041.3 2152.29  5048.7 2153.23
  5053.9 2151.56  5062.0 2153.68  5082.8 2156.72  5093.3 2157.20  5157.6 2164.81
#Mann=4,-1,0
  4810.9    0.07       0  4822.2    0.16       0  4987.0    0.07       0
  4991.0    0.16       0
Bank Sta=4987,4991
Exp/Cntr=0.3,0.1

Type RM Length L Ch R = 1,1194,47,47,47
BEGIN DESCRIPTION:
elmc515
END DESCRIPTION:
XS GIS Cut Line= 3
      1512567.43      6773552.41      1512750.77      6773529.63
      1512917.86      6773504.67
#Sta/Elev= 30
  4811.0 2163.70  4837.6 2161.36  4869.0 2159.40  4890.8 2156.85  4899.2 2155.13
  4909.3 2151.83  4919.4 2145.33  4929.5 2147.54  4939.6 2148.23  4959.7 2138.24
  4966.6 2132.22  4971.6 2134.71  4979.9 2126.11  4987.9 2122.79  4988.2 2122.29
  4991.7 2122.29  4991.9 2122.79  4995.4 2131.16  5000.4 2131.16  5010.1 2138.48
  5020.3 2142.54  5030.4 2145.18  5038.0 2145.71  5043.1 2147.55  5091.0 2151.45
  5101.1 2153.69  5112.3 2157.97  5131.5 2163.29  5141.6 2166.68  5164.7 2167.29
#Mann=4,-1,0
  4811.0    0.07       0  4837.6    0.16       0  4987.9    0.07       0
  4991.9    0.16       0
Bank Sta=4987.9,4991.9
Exp/Cntr=0.3,0.1

Type RM Length L Ch R = 1,1147,29,29,29
BEGIN DESCRIPTION:
elmc514
END DESCRIPTION:
XS GIS Cut Line= 3
      1512631.46      6773603.40      1512756.20      6773576.29
      1512896.21      6773526.36
#Sta/Elev= 30
  4871.5 2162.34  4876.8 2160.11  4915.7 2155.66  4920.8 2153.42  4926.3 2152.45
  4936.5 2149.94  4946.8 2148.16  4964.8 2146.91  4969.9 2141.99  4977.5 2139.26
  4987.7 2134.03  4996.0 2127.82  5001.2 2127.82  5004.1 2121.25  5004.3 2120.75
  5007.8 2120.75  5008.1 2121.25  5011.4 2123.02  5019.1 2131.00  5029.7 2136.06
  5036.9 2138.45  5061.6 2143.68  5067.7 2145.51  5073.0 2146.54  5098.5 2149.00
  5124.0 2152.40  5129.3 2155.65  5135.9 2157.85  5144.5 2161.13  5147.8 2161.13
#Mann=3,-1,0
  4871.5    0.16       0  5004.1    0.07       0  5008.1    0.16       0
Bank Sta=5004.1,5008.1
Exp/Cntr=0.3,0.1

Type RM Length L Ch R = 1,1118,46,46,46
BEGIN DESCRIPTION:
elmc513
END DESCRIPTION:
XS GIS Cut Line= 3
      1512661.80      6773668.52      1512771.39      6773600.16
      1512864.10      6773552.73
#Sta/Elev= 30
  4872.0 2160.48  4876.8 2160.48  4882.0 2158.28  4897.4 2156.67  4903.3 2156.53
  4924.5 2152.35  4934.0 2151.20  4946.5 2148.60  4955.2 2146.02  4961.1 2145.37
  4970.1 2142.10  4976.4 2138.97  4982.3 2137.68  4991.8 2131.41  4997.7 2126.60
  4998.3 2123.17  4998.6 2122.67  5002.1 2122.67  5002.3 2123.17  5006.0 2123.17
  5013.9 2130.07  5019.5 2133.92  5027.7 2137.21  5041.7 2140.85  5050.1 2143.44
  5058.3 2144.54  5072.6 2145.69  5080.5 2146.95  5102.7 2148.43  5105.3 2149.23
#Mann=3,-1,0
  4872.0    0.16       0  4998.3    0.07       0  5002.3    0.16       0
Bank Sta=4998.3,5002.3
Exp/Cntr=0.3,0.1

Type RM Length L Ch R = 1,1072,52,52,52
BEGIN DESCRIPTION:
elmc512
END DESCRIPTION:
XS GIS Cut Line= 3
      1512685.65      6773684.80      1512796.35      6773638.14
      1512871.12      6773589.00
#Sta/Elev= 30
  4876.7 2158.22  4879.0 2158.22  4881.4 2156.86  4886.8 2154.86  4897.7 2153.39
  4905.1 2151.21  4910.5 2151.89  4928.8 2149.98  4934.3 2150.60  4941.1 2148.88
  4952.0 2144.19  4958.0 2139.45  4963.4 2139.28  4973.7 2130.95  4979.7 2120.51
  4979.9 2120.01  4983.4 2120.01  4983.7 2120.51  4987.1 2121.56  4993.4 2132.01
  4999.0 2132.01  5003.7 2138.91  5009.7 2141.34  5024.8 2142.83  5031.1 2142.35
  5039.8 2142.51  5045.8 2142.94  5076.0 2145.68  5082.0 2146.77  5086.3 2146.97
#Mann=3,-1,0
  4876.7    0.16       0  4979.7    0.07       0  4983.7    0.16       0
Bank Sta=4979.7,4983.7
Exp/Cntr=0.3,0.1
