--- Elm 52.prj (project) ---

Proj Title=Elm 52 Base Level Engineering
Current Plan=p01
Default Exp/Contr=0.3,0.1
English Units
Geom File=g01
Flow File=f01
Plan File=p01
BEGIN DESCRIPTION:
Elm 52
END DESCRIPTION:

--- Elm 52.p01 (plan) ---

Plan Title=Multiple Run
Short Identifier=Multiple
Geom File=g01
Flow File=f01
Subcritical Flow
K Sum by GR= 0
Std Step Tol= 0.01
Critical Tol= 0.01
Num of Std Step Trials= 20
Max Error Tol= 0.3
Flow Tol Ratio= 0.001
Split Flow NTrial= 30
Split Flow Tol= 0.02
Split Flow Ratio= 0.02
Log Output Level= 0
Friction Slope Method= 1
Unsteady Friction Slope Method= 2
Unsteady Bridges Friction Slope Method= 1
Parabolic Critical Depth
Global Vel Dist=  1 , 1 , 1
Global Log Level= 0
CheckData=True
Encroach Param= -1, 0, 0, 0
BEGIN DESCRIPTION:
Multiple Run
END DESCRIPTION:

--- Elm 52.f01 (steady flow) ---

Flow Title=Multiple
Number of Profiles=7
Profile Names=10-year,25-year,50-year,1pct_min,100-year,1pct_plu,500-year
River Rch & RM= Elm 52,Reach-1,21995
     232     323     400     307     492     677     755
River Rch & RM= Elm 52,Reach-1,19836
     344     491     616     480     769    1060    1210
River Rch & RM= Elm 52,Reach-1,15251
     561     820    1050     826    1320    1820    2150
River Rch & RM= Elm 52,Reach-1,7211
     662     974    1250     991    1590    2190    2600
River Rch & RM= Elm 52,Reach-1,4534
     735    1090    1400    1110    1780    2450    2930
Boundary for River Rch & Prof#=Elm 52,Reach-1,1
Up Type=0
Dn Type=3
Dn Slope=0.005
Boundary for River Rch & Prof#=Elm 52,Reach-1,2
Up Type=0
Dn Type=3
Dn Slope=0.005
Boundary for River Rch & Prof#=Elm 52,Reach-1,3
Up Type=0
Dn Type=3
Dn Slope=0.005
Boundary for River Rch & Prof#=Elm 52,Reach-1,4
Up Type=0
Dn Type=3
Dn Slope=0.005
Boundary for River Rch & Prof#=Elm 52,Reach-1,5
Up Type=0
Dn Type=3
Dn Slope=0.005
Boundary for River Rch & Prof#=Elm 52,Reach-1,6
Up Type=0
Dn Type=3
Dn Slope=0.005
Boundary for River Rch & Prof#=Elm 52,Reach-1,7
Up Type=0
Dn Type=3
Dn Slope=0.005

--- Elm 52.g01 (geometry) ---

Geom Title=Existing Conditions

River Reach=Elm 52,Reach-1
Reach XY= 30
      1508305.00      6761938.00      1508713.00      6763544.39
      1509828.73      6764261.12      1510021.43      6764854.77
      1510647.20      6765181.79      1510691.36      6765574.56
      1511196.69      6765584.92      1511698.33      6764846.77
      1511997.38      6764931.50      1511906.88      6765432.31
      1512205.67      6765653.07      1512007.82      6766580.05
      1512647.20      6766931.79      1512465.02      6767498.05
      1512970.23      6767787.76      1513164.86      6767598.89
      1513348.83      6768180.14      1514407.43      6768543.52
      1514841.76      6769124.89      1515305.00      6769288.00
      1515277.70      6769561.90      1516288.73      6770220.79
      1516651.69      6770739.80      1516304.55      6771053.19
      1516712.67      6771794.52      1517301.48      6771839.45
      1516821.15      6772304.58      1517857.78      6772593.36
      1517763.95      6772844.67      1518055.00      6772938.00

Type RM Length L Ch R = 1,21995,154,154,154
BEGIN DESCRIPTION:
Elm 52 21995.025
END DESCRIPTION:
XS GIS Cut Line= 3
      1508193.58      6762149.84      1508348.81      6762086.13
      1508643.29      6761932.81
#Sta/Elev= 30
  4832.2 2352.74  4874.1 2350.02  4920.2 2345.38  4927.4 2343.92  4951.4 2342.25
  4956.8 2341.25  4974.3 2336.16  4980.8 2329.80  4986.2 2328.95  4995.2 2325.33
  5000.0 2325.33  5002.1 2324.15  5002.3 2323.65  5005.8 2323.65  5006.1 2324.15
  5018.2 2324.78  5026.2 2326.05  5031.8 2327.82  5048.3 2329.68  5092.5 2332.28
  5098.1 2331.92  5114.6 2333.10  5120.2 2332.80  5158.8 2334.91  5197.3 2340.13
  5203.0 2340.39  5232.5 2344.08  5255.0 2345.73  5307.8 2351.77  5332.0 2353.22
#Mann=3,-1,0
  4832.2    0.16       0  5002.1    0.07       0  5006.1    0.16       0
Bank Sta=5002.1,5006.1
Exp/Cntr=0.3,0.1

Type RM Length L Ch R = 1,21841,89,89,89
BEGIN DESCRIPTION:
Elm 52 21841.21
END DESCRIPTION:
XS GIS Cut Line= 3
      1508188.41      6762314.76      1508400.22      6762212.33
      1508631.40      6762041.53
#Sta/Elev= 30
  4758.8 2354.73  4767.3 2353.86  4789.8 2354.11  4812.4 2352.50  4874.7 2345.67
  4910.5 2343.06  4942.4 2338.50  4970.6 2333.45  4985.6 2327.86  4985.9 2327.36
  4989.6 2327.86  4993.2 2330.11  5008.0 2329.28  5014.2 2331.79  5028.8 2332.78
  5037.3 2331.82  5058.1 2331.81  5072.7 2332.89  5087.0 2331.69  5093.6 2329.20
  5099.8 2330.27  5158.3 2333.11  5179.2 2335.66  5193.8 2339.68  5229.3 2343.93
  5243.9 2347.17  5250.1 2347.17  5273.2 2350.48  5279.4 2350.09  5281.5 2351.83
#Mann=3,-1,0
  4758.8    0.16       0  4985.6    0.07       0  4989.6    0.16       0
Bank Sta=4985.6,4989.6
Exp/Cntr=0.3,0.1

Type RM Length L Ch R = 1,21752,90,90,90
BEGIN DESCRIPTION:
Elm 52 21752.1
END DESCRIPTION:
XS GIS Cut Line= 3
      1508221.45      6762361.62      1508445.36      6762285.24
      1508697.12      6762109.88
#Sta/Elev= 30
  4761.2 2352.94  4775.5 2352.39  4784.3 2351.39  4789.6 2351.58  4828.3 2346.33
  4883.6 2342.38  4909.7 2338.96  4934.0 2337.81  4946.3 2335.75  4965.7 2328.32
  4972.4 2324.07  4984.8 2323.49  4985.1 2322.99  4988.6 2322.99  4988.8 2323.49
  5046.1 2325.39  5053.2 2326.24  5118.6 2329.36  5139.6 2330.97  5160.5 2333.81
  5175.4 2338.49  5181.5 2339.03  5190.2 2341.44  5196.3 2342.00  5204.5 2344.26
  5232.1 2348.21  5240.8 2350.06  5246.9 2350.48  5261.8 2353.51  5304.6 2355.84
#Mann=3,-1,0
  4761.2    0.16       0  4984.8    0.07       0  4988.8    0.16       0
Bank Sta=4984.8,4988.8
Exp/Cntr=0.3,0.1

Type RM Length L Ch R = 1,21662,168,168,168
BEGIN DESCRIPTION:
Elm 52 21661.81
END DESCRIPTION:
XS GIS Cut Line= 3
      1508226.62      6762457.11      1508450.57      6762377.26
      1508707.50      6762193.23
#Sta/Elev= 30
  4754.5 2352.92  4784.6 2351.21  4805.9 2348.18  4837.7 2345.79  4854.9 2343.63
  4869.6 2343.31  4901.4 2340.17  4911.2 2338.30  4916.5 2338.77  4922.7 2337.28
  4947.3 2335.52  4972.8 2329.37  4978.1 2328.97  4992.0 2323.46  5001.7 2323.39
  5014.5 2321.63  5014.7 2321.13  5018.5 2321.63  5022.6 2322.30  5045.9 2321.86
  5102.4 2327.14  5131.9 2327.51  5159.0 2330.13  5173.7 2331.93  5188.4 2336.03
  5238.8 2345.76  5274.4 2350.72  5280.6 2352.89  5289.1 2354.46  5308.3 2355.93
#Mann=3,-1,0
  4754.5    0.16       0  5014.5    0.07       0  5018.5    0.16       0
Bank Sta=5014.5,5018.5
Exp/Cntr=0.3,0.1

Type RM Length L Ch R = 1,21494,92,92,92
BEGIN DESCRIPTION:
Elm 52 21493.5
END DESCRIPTION:
XS GIS Cut Line= 3
      1508327.31      6762615.10      1508507.86      6762524.83
      1508771.70      6762419.63
#Sta/Elev= 30
  4799.6 2341.90  4803.5 2340.32  4809.0 2340.66  4825.8 2336.74  4831.4 2338.35
  4848.2 2334.47  4853.8 2335.65  4870.5 2332.99  4876.1 2333.16  4886.5 2330.96
  4892.9 2328.77  4898.5 2329.28  4915.3 2326.92  4920.8 2327.11  4937.6 2325.37
  5001.5 2322.45  5027.3 2319.25  5027.6 2318.75  5031.3 2319.25  5052.2 2320.34
  5059.0 2322.08  5106.0 2323.45  5142.6 2326.39  5166.8 2333.22  5191.1 2339.08
  5196.5 2339.27  5220.7 2345.50  5250.4 2348.79  5267.5 2354.42  5285.5 2357.39
#Mann=3,-1,0
  4799.6    0.16       0  5027.3    0.07       0  5031.3    0.16       0
Bank Sta=5027.3,5031.3
Exp/Cntr=0.3,0.1

Type RM Length L Ch R = 1,21402,155,155,155
BEGIN DESCRIPTION:
Elm 52 21402.02
END DESCRIPTION:
XS GIS Cut Line= 3
      1508322.07      6762677.61      1508554.73      6762597.74
      1508799.69      6762542.93
#Sta/Elev= 30
  4746.5 2342.22  4763.1 2341.12  4789.0 2336.50  4794.3 2336.42  4820.3 2330.65
  4851.6 2327.65  4856.9 2328.09  4882.8 2325.85  4919.4 2324.28  4945.3 2322.09
  4976.6 2321.01  4982.2 2319.13  5009.2 2318.28  5009.4 2317.78  5012.9 2317.78
  5013.2 2318.28  5016.3 2318.52  5023.5 2320.56  5074.7 2321.11  5108.2 2323.75
  5146.5 2337.81  5151.6 2338.81  5156.7 2341.61  5177.2 2345.03  5187.5 2346.11
  5195.0 2348.92  5200.1 2349.14  5208.0 2351.94  5228.4 2355.78  5243.5 2357.24
#Mann=3,-1,0
  4746.5    0.16       0  5009.2    0.07       0  5013.2    0.16       0
Bank Sta=5009.2,5013.2
Exp/Cntr=0.3,0.1

Type RM Length L Ch R = 1,21247,200,200,200
BEGIN DESCRIPTION:
Elm 52 21246.98
END DESCRIPTION:
XS GIS Cut Line= 3
      1508356.80      6762760.94      1508599.87      6762736.63
      1508844.65      6762696.70
#Sta/Elev= 30
  4746.2 2337.72  4774.5 2332.80  4794.6 2328.14  4814.7 2324.88  4822.9 2324.35
  4827.9 2324.80  4834.8 2323.87  4875.0 2322.55  4945.4 2321.63  4965.5 2320.21
  4975.5 2318.46  4990.5 2317.90  5010.0 2315.97  5010.2 2315.47  5013.7 2315.47
  5014.0 2315.97  5017.0 2317.23  5026.1 2317.94  5073.4 2317.73  5078.5 2318.46
  5086.9 2318.29  5097.0 2319.81  5107.1 2325.25  5117.3 2333.47  5127.4 2339.25
  5134.9 2341.85  5147.7 2344.25  5167.9 2346.54  5208.5 2355.10  5238.5 2357.23
#Mann=3,-1,0
  4746.2    0.16       0  5010.0    0.07       0  5014.0    0.16       0
Bank Sta=5010,5014
Exp/Cntr=0.3,0.1

Type RM Length L Ch R = 1,21047,119,119,119
BEGIN DESCRIPTION:
Elm 52 21046.52
END DESCRIPTION:
XS GIS Cut Line= 3
      1508294.33      6762872.05      1508704.04      6762899.83
      1508850.83      6762868.74
#Sta/Elev= 30
  4587.6 2342.09  4628.4 2338.48  4648.4 2335.20  4658.4 2334.27  4698.5 2327.11
  4728.6 2323.31  4746.6 2322.00  4818.8 2319.08  4828.8 2319.30  4969.1 2315.68
  4979.2 2314.76  4987.2 2312.28  4987.4 2311.78  4990.9 2311.78  4991.2 2312.28
  4996.2 2314.51  5001.3 2314.51  5009.5 2319.96  5019.7 2325.50  5028.0 2331.08
  5033.1 2331.39  5050.3 2336.97  5060.6 2339.14  5070.8 2341.03  5082.8 2342.06
  5111.7 2346.49  5121.9 2348.60  5127.4 2350.97  5132.5 2351.08  5148.3 2354.48
#Mann=3,-1,0
  4587.6    0.16       0  4987.2    0.07       0  4991.2    0.16       0
Bank Sta=4987.2,4991.2
Exp/Cntr=0.3,0.1

Type RM Length L Ch R = 1,20928,187,187,187
BEGIN DESCRIPTION:
Elm 52 20928.46
END DESCRIPTION:
XS GIS Cut Line= 3
      1508278.68      6762944.96      1508646.75      6762986.63
      1508839.45      6762969.27
#Sta/Elev= 30
  4626.6 2339.56  4643.0 2339.34  4698.2 2333.79  4713.5 2330.64  4723.5 2329.18
  4733.6 2328.45  4763.8 2323.83  4804.0 2320.97  4859.8 2318.75  4924.8 2316.94
  4955.0 2315.66  4965.7 2314.44  4975.1 2313.75  5003.3 2313.46  5003.6 2312.96
  5007.1 2312.96  5007.3 2313.46  5015.3 2314.96  5039.0 2316.36  5055.5 2319.87
  5065.5 2322.70  5095.7 2329.13  5105.7 2332.65  5125.8 2337.49  5144.9 2340.72
  5149.9 2340.89  5166.0 2343.31  5176.0 2345.30  5185.8 2346.63  5190.5 2346.63
#Mann=5,-1,0
  4626.6    0.16       0  4859.8    0.07       0  4965.7    0.16       0
  5003.3    0.07       0  5007.3    0.16       0
Bank Sta=5003.3,5007.3
Exp/Cntr=0.3,0.1

Type RM Length L Ch R = 1,20741,220,220,220
BEGIN DESCRIPTION:
Elm 52 20741.35
END DESCRIPTION:
XS GIS Cut Line= 3
      1508327.32      6763172.39      1508610.29      6763158.51
      1508835.93      6763108.17
#Sta/Elev= 30
  4722.4 2339.56  4730.1 2338.52  4760.1 2336.11  4780.1 2333.31  4800.2 2329.66
  4850.2 2319.24  4880.3 2316.61  4900.2 2316.32  4909.7 2316.14  4914.7 2316.59
  4960.4 2315.09  4980.4 2312.92  4988.4 2310.87  4988.7 2310.37  4992.2 2310.37
  4992.4 2310.87  5020.8 2311.72  5028.5 2313.02  5033.6 2313.28  5051.2 2313.12
  5092.5 2313.75  5125.6 2315.62  5143.7 2317.64  5169.1 2322.52  5174.5 2324.85
  5205.2 2334.44  5212.5 2336.18  5225.7 2338.10  5233.9 2339.97  5236.9 2339.97
#Mann=5,-1,0
  4722.4    0.16       0  4900.2    0.07       0  4988.4    0.07       0
  4992.4    0.07       0  5051.2    0.16       0
Bank Sta=4988.4,4992.4
Exp/Cntr=0.3,0.1

Type RM Length L Ch R = 1,20521,147,147,147
BEGIN DESCRIPTION:
Elm 52 20521.471
END DESCRIPTION:
XS GIS Cut Line= 3
      1508354.99      6763488.01      1508654.99      6763363.01
      1508954.98      6763188.01
#Sta/Elev= 30
  4675.0 2341.30  4684.2 2339.25  4713.5 2335.58  4720.8 2335.43  4742.7 2334.35
  4761.1 2331.63  4766.6 2331.74  4790.4 2326.89  4808.8 2324.74  4819.6 2323.98
  4826.7 2321.88  4837.5 2320.58  4843.5 2318.27  4848.9 2318.38  4867.3 2315.31
  4880.8 2315.43  4920.4 2312.43  4967.5 2311.55  5000.9 2308.93  5001.2 2308.43
  5004.9 2308.93  5049.7 2311.08  5114.5 2311.85  5150.5 2313.97  5166.2 2316.02
  5179.0 2317.75  5200.5 2323.57  5222.0 2331.70  5237.8 2335.99  5347.3 2351.00
#Mann=7,-1,0
  4675.0    0.16       0  4720.8   0.035       0  4808.8    0.16       0
  5000.9    0.07       0  5004.9    0.16       0  5049.7    0.07       0
  5166.2    0.16       0
Bank Sta=5000.9,5004.9
Exp/Cntr=0.3,0.1

Type RM Length L Ch R = 1,20374,136,136,136
BEGIN DESCRIPTION:
Elm 52 20373.7
END DESCRIPTION:
XS GIS Cut Line= 3
      1508516.58      6763583.83      1508702.30      6763495.31
      1508897.59      6763312.12
#Sta/Elev= 30
  4796.0 2324.48  4805.3 2322.53  4821.6 2321.01  4827.5 2319.79  4844.3 2317.90
  4882.9 2315.04  4895.2 2313.07  4926.8 2311.61  4963.3 2309.73  4971.5 2307.86
  4984.0 2306.82  4984.2 2306.32  4987.7 2306.32  4988.0 2306.82  4993.6 2308.70
  5000.5 2309.41  5044.3 2309.00  5076.5 2309.63  5093.7 2309.92  5128.7 2308.91
  5150.3 2309.02  5178.7 2311.99  5192.8 2311.96  5199.7 2312.89  5215.6 2316.45
  5221.2 2318.43  5235.3 2325.45  5249.5 2330.81  5263.7 2335.00  5269.5 2335.50
#Mann=7,-1,0
  4796.0   0.035       0  4926.8    0.07       0  4984.0    0.07       0
  4988.0    0.07       0  5076.5   0.035       0  5128.7    0.07       0
  5215.6    0.16       0
Bank Sta=4984,4988
Exp/Cntr=0.3,0.1

Type RM Length L Ch R = 1,20238,103,103,103
BEGIN DESCRIPTION:
Elm 52 20238.27
END DESCRIPTION:
XS GIS Cut Line= 3
      1508648.50      6763773.06      1508778.69      6763592.53
      1508947.12      6763365.07
#Sta/Elev= 30
  4772.0 2317.23  4788.0 2316.05  4794.2 2314.92  4808.9 2314.70  4815.2 2313.83
  4865.4 2312.32  4930.4 2311.45  4959.8 2309.49  4980.7 2307.35  4985.8 2305.93
  4986.1 2305.43  4989.6 2305.43  4989.8 2305.93  5010.0 2306.51  5030.9 2306.24
  5045.5 2307.27  5056.6 2307.40  5074.7 2307.45  5116.4 2306.00  5151.9 2306.50
  5166.5 2307.41  5174.8 2309.68  5186.7 2311.86  5210.4 2313.11  5231.2 2320.78
  5237.4 2324.07  5252.1 2329.86  5260.5 2332.54  5272.6 2334.24  5277.6 2334.24
#Mann=6,-1,0
  4772.0    0.07       0  4985.8    0.07       0  4989.8    0.07       0
  5056.6   0.035       0  5174.8    0.07       0  5186.7    0.16       0
Bank Sta=4985.8,4989.8
Exp/Cntr=0.3,0.1

Type RM Length L Ch R = 1,20135,129,129,129
BEGIN DESCRIPTION:
Elm 52 20134.76
END DESCRIPTION:
XS GIS Cut Line= 3
      1508730.06      6763800.89      1508882.86      6763592.53
      1509013.06      6763408.52
#Sta/Elev= 30
  4737.2 2312.17  4756.7 2311.58  4764.7 2311.88  4842.4 2310.15  4871.7 2310.47
  4877.9 2310.02  4922.8 2309.91  4942.7 2309.13  4951.2 2308.19  4957.4 2308.34
  4986.7 2305.27  4992.9 2305.34  4993.3 2304.13  4993.5 2303.63  4997.0 2303.63
  4997.3 2304.13  5013.7 2304.29  5022.4 2305.02  5072.9 2305.68  5079.0 2305.29
  5086.9 2305.85  5114.7 2311.48  5123.3 2312.55  5150.4 2313.94  5165.1 2320.45
  5169.8 2323.42  5172.6 2325.19  5179.9 2327.73  5194.7 2331.26  5221.0 2334.80
#Mann=6,-1,0
  4737.2    0.16       0  4764.7    0.07       0  4922.8   0.035       0
  4993.3   0.035       0  4997.3   0.035       0  5169.8    0.16       0
Bank Sta=4993.3,4997.3
Exp/Cntr=0.3,0.1

Type RM Length L Ch R = 1,20006,170,170,170
BEGIN DESCRIPTION:
Elm 52 20005.73
END DESCRIPTION:
XS GIS Cut Line= 3
      1508728.37      6763830.36      1508993.97      6763637.67
      1509150.12      6763453.76
#Sta/Elev= 30
  4660.7 2312.79  4688.8 2311.37  4723.5 2310.86  4789.4 2309.04  4795.5 2309.68
  4804.0 2308.93  4821.6 2308.93  4931.6 2307.42  4996.6 2304.21  5015.4 2300.81
  5015.7 2300.31  5019.2 2300.31  5019.4 2300.81  5039.4 2304.16  5057.5 2310.13
  5067.1 2313.17  5074.5 2313.68  5081.1 2313.08  5095.4 2313.31  5103.1 2314.35
  5109.7 2313.86  5117.4 2314.78  5187.7 2316.49  5195.4 2319.18  5201.9 2318.85
  5209.7 2322.03  5216.2 2321.46  5223.9 2324.86  5228.6 2324.40  5230.1 2324.25
#Mann=7,-1,0
  4660.7    0.16       0  4723.5    0.07       0  4821.6   0.035       0
  5015.4   0.035       0  5019.4   0.035       0  5057.5    0.07       0
  5228.6   0.035       0
Bank Sta=5015.4,5019.4
Exp/Cntr=0.3,0.1

Type RM Length L Ch R = 1,19836,93,93,93
BEGIN DESCRIPTION:
Elm 52 19836.06
END DESCRIPTION:
XS GIS Cut Line= 3
      1508971.39      6763889.42      1509106.82      6763738.37
      1509294.35      6763580.35
#Sta/Elev= 30
  4792.6 2306.05  4817.6 2304.77  4864.4 2303.55  4902.0 2301.55  4923.7 2301.54
  4930.4 2300.75  4952.1 2300.23  4958.8 2299.20  4966.3 2299.26  4973.1 2298.33
  4980.5 2298.48  4987.3 2296.99  4997.6 2297.69  4999.7 2296.78  5000.0 2296.28
  5003.5 2296.28  5003.7 2296.78  5016.0 2298.23  5030.3 2302.89  5051.2 2306.50
  5058.5 2306.22  5086.3 2308.64  5129.2 2310.22  5150.0 2309.98  5157.8 2309.24
  5164.3 2310.47  5172.1 2309.32  5178.6 2309.90  5186.4 2308.72  5240.7 2311.85
#Mann=4,-1,0
  4792.6   0.035       0  4864.4    0.07       0  4999.7    0.07       0
  5003.7    0.07       0
Bank Sta=4999.7,5003.7
Exp/Cntr=0.3,0.1

Type RM Length L Ch R = 1,19743,147,147,147
BEGIN DESCRIPTION:
Elm 52 19742.62
END DESCRIPTION:
XS GIS Cut Line= 3
      1509000.94      6763927.58      1509158.90      6763811.28
      1509320.14      6763726.33
#Sta/Elev= 30
  4809.0 2307.54  4833.1 2306.58  4847.8 2305.14  4861.1 2304.51  4868.6 2303.89
  4889.5 2304.17  4904.1 2303.35  4925.8 2300.24  4948.0 2299.00  4962.7 2299.48
  4975.5 2300.72  4989.7 2300.34  4998.2 2299.04  5010.0 2298.45  5010.3 2297.95
  5013.8 2297.95  5014.0 2298.45  5034.7 2301.47  5042.3 2301.22  5048.0 2302.19
  5056.8 2301.66  5064.4 2301.78  5070.0 2302.79  5086.4 2303.21  5092.1 2304.25
  5108.4 2304.29  5114.1 2305.20  5146.8 2305.99  5152.5 2306.64  5187.4 2307.77
#Mann=5,-1,0
  4809.0   0.035       0  4861.1    0.07       0  5010.0    0.07       0
  5014.0    0.07       0  5056.8    0.16       0
Bank Sta=5010,5014
Exp/Cntr=0.3,0.1

Type RM Length L Ch R = 1,19596,144,144,144
BEGIN DESCRIPTION:
Elm 52 19596.18
END DESCRIPTION:
XS GIS Cut Line= 3
      1509162.38      6764043.91      1509230.08      6763911.98
      1509342.92      6763743.58
#Sta/Elev= 30
  4852.5 2307.06  4867.0 2306.06  4872.6 2305.89  4894.8 2304.07  4926.6 2302.38
  4939.2 2300.70  4955.7 2299.30  4961.4 2299.14  4971.5 2297.52  4977.9 2293.18
  4992.0 2292.07  4992.3 2291.57  4995.8 2291.57  4996.0 2292.07  5000.1 2293.48
  5006.2 2293.78  5015.1 2295.07  5021.1 2295.54  5029.7 2296.75  5036.1 2298.23
  5042.1 2299.03  5057.1 2300.83  5073.8 2302.18  5108.2 2303.46  5114.2 2304.08
  5144.2 2305.14  5159.2 2305.97  5186.2 2306.72  5195.2 2307.40  5203.5 2307.68
#Mann=4,-1,0
  4852.5    0.07       0  4992.0    0.07       0  4996.0    0.07       0
  5073.8    0.16       0
Bank Sta=4992,4996
Exp/Cntr=0.3,0.1

Type RM Length L Ch R = 1,19452,99,99,99
BEGIN DESCRIPTION:
Elm 52 19451.67
END DESCRIPTION:
XS GIS Cut Line= 3
      1509308.19      6764103.00      1509365.50      6763944.97
      1509434.36      6763791.73
#Sta/Elev= 30
  4835.8 2305.64  4851.8 2304.45  4883.7 2303.19  4894.3 2302.27  4899.7 2301.21
  4930.3 2299.09  4947.5 2296.81  4960.9 2293.91  4968.8 2291.81  4979.4 2291.08
  4984.2 2290.31  4984.5 2289.81  4988.0 2289.81  4988.2 2290.31  5003.9 2290.85
  5005.3 2291.61  5010.5 2294.44  5016.0 2295.77  5022.5 2299.90  5055.4 2301.29
  5067.8 2302.45  5090.9 2303.16  5108.6 2304.38  5114.1 2304.09  5131.8 2305.16
  5137.2 2305.07  5154.1 2305.83  5160.4 2306.92  5165.9 2306.79  5171.9 2307.27
#Mann=4,-1,0
  4835.8    0.07       0  4984.2    0.07       0  4988.2    0.07       0
  5005.3    0.16       0
Bank Sta=4984.2,4988.2
Exp/Cntr=0.3,0.1

Type RM Length L Ch R = 1,19353,121,121,121
BEGIN DESCRIPTION:
Elm 52 19352.65
END DESCRIPTION:
XS GIS Cut Line= 3
      1509407.16      6764148.08      1509448.83      6763991.84
      1509514.81      6763795.64
#Sta/Elev= 30
  4834.9 2304.47  4837.5 2304.47  4848.2 2302.98  4883.1 2301.21  4888.3 2300.15
  4897.1 2299.35  4923.2 2297.66  4928.4 2297.70  4938.5 2295.91  4958.2 2293.92
  4967.8 2291.76  4969.5 2291.36  4990.2 2290.61  5001.1 2289.21  5001.4 2288.71
  5004.9 2288.71  5005.1 2289.21  5011.2 2293.58  5021.8 2297.66  5029.3 2297.82
  5053.4 2299.77  5066.1 2300.11  5097.6 2302.06  5123.9 2304.28  5129.1 2304.22
  5148.4 2305.69  5169.5 2308.48  5180.0 2308.52  5199.7 2310.31  5203.6 2310.31
#Mann=4,-1,0
  4834.9    0.07       0  4967.8    0.16       0  5001.1    0.07       0
  5005.1    0.16       0
Bank Sta=5001.1,5005.1
Exp/Cntr=0.3,0.1

Type RM Length L Ch R = 1,19232,149,149,149
BEGIN DESCRIPTION:
Elm 52 19232.08
END DESCRIPTION:
XS GIS Cut Line= 3
      1509426.26      6764168.93      1509559.94      6764028.30
      1509639.36      6763902.26
#Sta/Elev= 30
  4811.6 2304.46  4825.7 2303.26  4839.8 2302.62  4854.0 2302.52  4868.1 2299.51
  4871.3 2299.44  4875.0 2299.35  4896.1 2297.19  4910.2 2296.90  4917.5 2296.17
  4931.7 2295.81  4945.8 2294.02  4960.0 2291.30  4981.0 2289.07  4993.2 2286.59
  4993.4 2286.09  4996.9 2286.09  4997.2 2286.59  5005.6 2286.64  5024.1 2294.95
  5039.4 2297.54  5060.6 2299.40  5081.8 2300.74  5097.1 2303.02  5103.0 2304.47
  5112.4 2305.25  5118.3 2306.79  5133.6 2307.71  5139.5 2309.03  5154.6 2310.60
#Mann=4,-1,0
  4811.6    0.07       0  4871.3    0.16       0  4993.2    0.07       0
  4997.2    0.16       0
Bank Sta=4993.2,4997.2
Exp/Cntr=0.3,0.1

Type RM Length L Ch R = 1,19083,110,110,110
BEGIN DESCRIPTION:
Elm 52 19082.999
END DESCRIPTION:
XS GIS Cut Line= 3
      1509505.04      6764187.98      1509649.08      6764130.99
      1509854.99      6763838.02
#Sta/Elev= 30
  4845.1 2302.46  4859.9 2300.85  4866.6 2299.00  4889.6 2296.80  4909.9 2295.86
  4943.7 2294.78  4984.9 2286.89  5000.0 2287.30  5014.9 2286.81  5018.5 2286.60
  5018.7 2286.10  5022.2 2286.10  5022.5 2286.60  5028.1 2287.26  5041.4 2292.82
  5056.2 2296.39  5077.1 2297.46  5106.8 2300.32  5127.7 2303.17  5136.4 2303.17
  5157.3 2306.80  5172.1 2308.05  5193.0 2311.31  5243.5 2314.67  5264.5 2317.44
  5300.2 2323.46  5315.0 2326.46  5321.5 2329.55  5329.8 2331.37  5358.1 2334.71
#Mann=5,-1,0
  4845.1    0.16       0  4909.9    0.07       0  5014.9    0.16       0
  5018.5    0.07       0  5022.5    0.16       0
Bank Sta=5018.5,5022.5
Exp/Cntr=0.3,0.1

Type RM Length L Ch R = 1,18973,88,88,88
BEGIN DESCRIPTION:
Elm 52 18972.83
END DESCRIPTION:
XS GIS Cut Line= 3
      1509592.93      6764325.17      1509738.76      6764188.02
      1509900.09      6763986.79
#Sta/Elev= 30
  4801.0 2301.41  4814.7 2299.73  4843.1 2297.64  4857.2 2295.68  4892.4 2293.51
  4899.7 2292.29  4934.9 2290.47  4954.1 2287.69  4963.2 2285.74  4984.2 2284.99
  4989.5 2284.06  4989.8 2283.56  4993.3 2283.56  4993.5 2284.06  4997.6 2285.14
  5001.2 2285.14  5005.4 2287.97  5013.4 2290.54  5034.2 2294.74  5048.6 2295.97
  5063.0 2296.30  5069.4 2297.44  5098.2 2299.90  5155.0 2307.41  5162.2 2307.80
  5168.6 2309.10  5232.7 2314.80  5247.1 2315.65  5255.0 2316.80  5259.1 2317.92
#Mann=4,-1,0
  4801.0    0.07       0  4954.1    0.16       0  4989.5    0.07       0
  4993.5    0.16       0
Bank Sta=4989.5,4993.5
Exp/Cntr=0.3,0.1

Type RM Length L Ch R = 1,18885,124,124,124
BEGIN DESCRIPTION:
Elm 52 18885.05
END DESCRIPTION:
XS GIS Cut Line= 3
      1509599.86      6764340.80      1509809.94      6764238.37
      1509954.07      6764099.45
#Sta/Elev= 30
  4769.9 2301.53  4775.6 2300.50  4807.0 2297.33  4812.5 2297.32  4829.5 2295.15
  4842.4 2294.53  4874.6 2291.61  4900.3 2290.25  4925.2 2288.08  4931.4 2286.34
  4947.7 2284.52  4973.9 2283.09  4974.1 2282.59  4977.6 2282.59  4977.9 2283.09
  4987.0 2285.83  4998.3 2291.35  5003.6 2291.35  5014.5 2293.25  5021.7 2293.19
  5056.9 2295.92  5071.1 2298.12  5085.2 2299.17  5092.4 2300.18  5106.6 2303.17
  5113.5 2303.90  5127.7 2306.70  5141.8 2306.84  5149.0 2307.77  5203.8 2311.94
#Mann=4,-1,0
  4769.9    0.07       0  4900.3    0.16       0  4973.9    0.07       0
  4977.9    0.16       0
Bank Sta=4973.9,4977.9
Exp/Cntr=0.3,0.1

Type RM Length L Ch R = 1,18761,97,97,97
BEGIN DESCRIPTION:
Elm 52 18761.21
END DESCRIPTION:
XS GIS Cut Line= 3
      1509672.80      6764464.06      1509858.55      6764347.74
      1510091.42      6764216.65
#Sta/Elev= 30
  4774.4 2298.64  4837.4 2294.78  4858.4 2294.17  4873.9 2293.29  4925.8 2292.32
  4954.0 2289.99  4977.6 2284.94  4983.6 2282.57  4986.6 2280.31  4986.9 2279.81
  4990.4 2279.81  4990.6 2280.31  5020.9 2282.44  5026.6 2284.13  5035.4 2285.70
  5042.6 2286.08  5048.3 2287.60  5058.3 2287.87  5064.2 2289.95  5085.9 2294.21
  5092.8 2297.07  5101.8 2298.52  5107.6 2298.56  5123.5 2302.53  5129.2 2302.78
  5145.2 2305.37  5182.8 2306.97  5210.2 2309.15  5253.5 2311.32  5260.8 2312.33
#Mann=4,-1,0
  4774.4    0.07       0  4858.4    0.16       0  4986.6    0.07       0
  4990.6    0.16       0
Bank Sta=4986.6,4990.6
Exp/Cntr=0.3,0.1

Type RM Length L Ch R = 1,18664,111,111,111
BEGIN DESCRIPTION:
Elm 52 18664.25
END DESCRIPTION:
XS GIS Cut Line= 3
      1509731.85      6764533.49      1509919.32      6764424.13
      1510096.37      6764278.32
#Sta/Elev= 30
  4766.9 2296.68  4803.0 2294.98  4809.3 2294.99  4825.0 2294.14  4862.2 2294.19
  4868.0 2293.76  4920.9 2292.68  4955.8 2291.10  4969.7 2289.45  4983.9 2286.45
  4991.7 2282.59  4999.6 2279.10  5004.1 2278.11  5004.3 2277.61  5007.8 2277.61
  5008.1 2278.11  5013.9 2278.78  5020.4 2280.31  5028.3 2281.21  5042.6 2287.48
  5049.1 2290.04  5063.5 2297.19  5069.9 2298.72  5084.3 2300.75  5098.6 2301.96
  5162.5 2305.76  5191.1 2308.23  5205.5 2308.65  5209.6 2309.31  5213.3 2309.31
#Mann=4,-1,0
  4766.9    0.07       0  4803.0    0.16       0  5004.1    0.07       0
  5008.1    0.16       0
Bank Sta=5004.1,5008.1
Exp/Cntr=0.3,0.1

Type RM Length L Ch R = 1,18553,94,94,94
BEGIN DESCRIPTION:
Elm 52 18553.42
END DESCRIPTION:
XS GIS Cut Line= 3
      1509801.29      6764580.37      1510007.86      6764495.31
      1510113.76      6764417.18
#Sta/Elev= 30
  4781.6 2292.58  4796.0 2292.25  4818.1 2292.18  4825.3 2291.81  4830.7 2292.11
  4839.7 2291.74  4872.1 2291.53  4908.0 2290.50  4931.9 2287.96  4937.3 2288.00
  4955.9 2284.50  4961.3 2284.61  4969.5 2282.74  4979.8 2279.18  4983.2 2278.29
  4983.5 2277.79  4987.0 2277.79  4987.2 2278.29  4991.1 2279.30  5000.7 2286.27
  5005.0 2286.27  5008.3 2291.39  5029.1 2292.98  5037.5 2293.97  5051.1 2296.36
  5064.6 2298.28  5087.7 2300.24  5100.9 2301.83  5114.7 2302.99  5136.6 2304.10
#Mann=3,-1,0
  4781.6    0.16       0  4983.2    0.07       0  4987.2    0.16       0
Bank Sta=4983.2,4987.2
Exp/Cntr=0.3,0.1

Type RM Length L Ch R = 1,18459,120,120,120
BEGIN DESCRIPTION:
Elm 52 18459.35
END DESCRIPTION:
XS GIS Cut Line= 3
      1509844.68      6764615.10      1510007.86      6764590.80
      1510115.51      6764543.92
#Sta/Elev= 30
  4837.6 2291.13  4847.4 2290.87  4852.5 2291.27  4878.4 2290.56  4898.6 2289.56
  4908.7 2289.53  4916.8 2288.65  4921.8 2289.11  4949.1 2285.64  4959.2 2282.64
  4969.4 2280.31  4979.5 2280.66  4986.1 2278.08  4991.1 2277.93  4998.6 2276.38
  5002.6 2276.38  5008.4 2275.57  5008.6 2275.07  5012.1 2275.07  5012.4 2275.57
  5019.0 2283.46  5024.4 2285.43  5032.2 2287.25  5042.4 2288.79  5047.9 2288.85
  5054.0 2289.92  5076.7 2292.18  5086.7 2292.48  5108.5 2295.34  5120.0 2295.36
#Mann=3,-1,0
  4837.6    0.16       0  5008.4    0.07       0  5012.4    0.16       0
Bank Sta=5008.4,5012.4
Exp/Cntr=0.3,0.1

Type RM Length L Ch R = 1,18339,125,125,125
BEGIN DESCRIPTION:
Elm 52 18339.14
END DESCRIPTION:
XS GIS Cut Line= 3
      1509825.57      6764722.74      1510002.65      6764712.33
      1510131.44      6764660.81
#Sta/Elev= 30
  4820.1 2299.96  4829.6 2299.29  4839.6 2297.55  4849.6 2295.01  4869.6 2291.92
  4879.6 2290.61  4889.7 2290.21  4899.7 2288.11  4929.7 2283.00  4939.7 2279.84
  4949.8 2277.62  4959.8 2277.80  4969.8 2275.52  4977.8 2271.22  4978.1 2270.72
  4981.6 2270.72  4981.8 2271.22  4985.4 2274.52  4990.4 2274.39  4996.2 2275.78
  5001.4 2275.78  5010.8 2280.97  5019.4 2286.64  5032.3 2287.15  5049.0 2289.04
  5078.6 2288.66  5086.2 2288.87  5102.9 2290.24  5108.2 2289.94  5136.2 2291.75
#Mann=3,-1,0
  4820.1    0.16       0  4977.8    0.07       0  4981.8    0.16       0
Bank Sta=4977.8,4981.8
Exp/Cntr=0.3,0.1

Type RM Length L Ch R = 1,18214,98,98,98
BEGIN DESCRIPTION:
Elm 52 18213.73
END DESCRIPTION:
XS GIS Cut Line= 3
      1509827.32      6764894.61      1510011.33      6764835.59
      1510148.51      6764740.08
#Sta/Elev= 30
  4809.7 2305.66  4813.7 2304.75  4819.0 2305.17  4845.9 2302.84  4861.5 2302.62
  4898.2 2299.20  4910.1 2297.45  4922.8 2294.71  4947.5 2293.31  4954.3 2289.83
  4964.8 2283.35  4974.4 2275.45  4979.6 2274.07  4985.8 2272.65  4996.3 2273.62
  5002.2 2272.13  5017.2 2271.06  5017.5 2270.56  5021.0 2270.56  5021.2 2271.06
  5025.3 2272.07  5031.8 2277.30  5040.2 2281.56  5046.3 2285.29  5090.8 2288.30
  5117.8 2288.79  5132.7 2289.89  5147.5 2290.09  5153.6 2290.62  5170.1 2290.76
#Mann=5,-1,0
  4809.7    0.16       0  4861.5    0.07       0  4898.2    0.16       0
  5017.2    0.07       0  5021.2    0.16       0
Bank Sta=5017.2,5021.2
Exp/Cntr=0.3,0.1

Type RM Length L Ch R = 1,18116,108,108,108
BEGIN DESCRIPTION:
Elm 52 18115.83
END DESCRIPTION:
XS GIS Cut Line= 3
      1509955.02      6764937.99      1510074.78      6764908.22
      1510154.99      6764838.01
#Sta/Elev= 30
  4876.6 2296.67  4879.2 2296.67  4886.9 2294.79  4894.7 2293.54  4899.8 2293.66
  4907.5 2292.92  4941.2 2292.18  4948.7 2287.90  4959.0 2282.40  4969.3 2277.48
  4977.3 2274.45  4982.5 2269.98  4987.9 2269.24  4988.2 2268.74  4991.7 2268.74
  4991.9 2269.24  4997.5 2269.97  4999.3 2269.97  5003.5 2269.97  5007.4 2270.51
  5014.1 2270.85  5021.7 2272.38  5028.3 2274.59  5035.9 2276.86  5056.8 2286.25
  5078.6 2287.16  5085.3 2288.05  5092.9 2288.10  5099.5 2288.49  5106.6 2288.26
#Mann=4,-1,0
  4876.6    0.07       0  4987.9    0.07       0  4991.9    0.07       0
  4999.3    0.16       0
Bank Sta=4987.9,4991.9
Exp/Cntr=0.3,0.1

Type RM Length L Ch R = 1,18008,101,101,101
BEGIN DESCRIPTION:
Elm 52 18008.38
END DESCRIPTION:
XS GIS Cut Line= 3
      1509973.13      6765092.54      1510150.22      6764984.90
      1510245.70      6764856.43
#Sta/Elev= 30
  4792.0 2292.79  4811.0 2292.33  4826.5 2291.47  4832.4 2291.69  4869.2 2291.06
  4876.1 2290.55  4884.7 2288.82  4890.5 2290.18  4906.0 2289.33  4921.5 2289.13
  4927.3 2288.26  4948.6 2286.62  4958.0 2284.48  4964.1 2280.99  4979.6 2276.39
  4990.8 2271.15  4993.1 2270.18  4997.0 2267.12  4997.3 2266.62  5000.9 2266.62
  5001.2 2267.12  5007.8 2267.20  5014.8 2268.05  5021.1 2268.19  5029.5 2270.45
  5035.7 2271.19  5050.3 2274.67  5071.1 2284.57  5107.5 2286.49  5159.3 2287.23
#Mann=4,-1,0
  4792.0    0.07       0  4990.8    0.16       0  4997.0    0.07       0
  5001.2    0.16       0
Bank Sta=4997,5001.2
Exp/Cntr=0.3,0.1

Type RM Length L Ch R = 1,17907,111,111,111
BEGIN DESCRIPTION:
Elm 52 17907.22
END DESCRIPTION:
XS GIS Cut Line= 3
      1510164.12      6765187.99      1510230.08      6765045.66
      1510276.60      6764871.64
#Sta/Elev= 30
  4835.2 2292.62  4867.9 2292.00  4874.1 2291.42  4890.3 2291.21  4896.3 2290.64
  4912.3 2290.46  4924.7 2289.79  4947.6 2289.24  4970.5 2287.42  4978.5 2284.69
  4987.9 2275.35  4992.0 2272.34  5000.0 2267.01  5008.2 2265.13  5008.5 2264.63
  5012.1 2264.63  5012.4 2265.13  5020.7 2266.22  5033.4 2270.25  5041.4 2270.12
  5051.8 2271.93  5062.1 2277.27  5068.2 2282.00  5073.4 2283.53  5093.2 2284.51
  5124.2 2285.06  5143.2 2285.95  5148.4 2285.43  5155.3 2285.32  5172.2 2286.23
#Mann=4,-1,0
  4835.2    0.07       0  4874.1    0.16       0  5008.2    0.07       0
  5012.4    0.16       0
Bank Sta=5008.2,5012.4
Exp/Cntr=0.3,0.1

Type RM Length L Ch R = 1,17796,100,100,100
BEGIN DESCRIPTION:
Elm 52 17795.99
END DESCRIPTION:
XS GIS Cut Line= 3
      1510252.64      6765210.61      1510344.66      6765036.98
      1510386.27      6764842.80
#Sta/Elev= 30
  4806.5 2290.84  4840.7 2290.09  4890.3 2288.13  4906.6 2288.18  4912.3 2286.89
  4922.6 2286.79  4928.6 2285.91  4934.3 2284.52  4945.0 2278.17  4950.6 2275.58
  4956.6 2271.17  4967.0 2266.04  4972.6 2264.98  4977.1 2262.89  4977.4 2262.39
  4981.1 2262.39  4981.3 2262.89  4989.0 2263.83  4999.6 2267.92  5012.2 2268.38
  5022.4 2269.50  5028.0 2275.44  5033.1 2275.52  5042.9 2280.91  5053.1 2281.86
  5072.3 2282.50  5083.8 2281.84  5104.2 2283.04  5114.5 2282.09  5201.6 2289.20
#Mann=3,-1,0
  4806.5    0.16       0  4977.1    0.07       0  4981.3    0.16       0
Bank Sta=4977.1,4981.3
Exp/Cntr=0.3,0.1

Type RM Length L Ch R = 1,17696,55,55,55
BEGIN DESCRIPTION:
Elm 52 17695.83
END DESCRIPTION:
XS GIS Cut Line= 3
      1510322.07      6765252.29      1510424.52      6765097.74
      1510483.57      6764908.46
#Sta/Elev= 30
  4803.4 2288.88  4816.1 2288.91  4822.1 2287.60  4852.2 2286.68  4858.2 2285.42
  4873.3 2284.60  4903.4 2284.10  4945.5 2282.23  4960.5 2277.92  4975.6 2271.55
  4981.6 2270.62  4985.7 2265.97  4991.3 2265.97  4996.9 2262.69  4997.2 2262.19
  5001.1 2262.69  5005.7 2264.46  5011.0 2264.15  5030.5 2266.05  5038.2 2270.78
  5043.5 2269.25  5051.4 2273.30  5070.7 2277.28  5076.0 2277.65  5082.8 2279.27
  5108.5 2281.61  5114.3 2283.15  5141.0 2286.82  5146.2 2288.48  5187.1 2293.59
#Mann=3,-1,0
  4803.4    0.16       0  4996.9    0.07       0  5001.1    0.16       0
Bank Sta=4996.9,5001.1
Exp/Cntr=0.3,0.1

Type RM Length L Ch R = 1,17641,129,129,129
BEGIN DESCRIPTION:
Elm 52 17641.327
END DESCRIPTION:
XS GIS Cut Line= 3
      1510454.99      6765188.03      1510482.33      6765088.42
      1510555.03      6764987.96
#Sta/Elev= 30
  4896.7 2281.39  4914.0 2281.26  4938.2 2278.21  4948.4 2273.68  4953.6 2272.92
  4959.0 2268.81  4969.3 2267.55  4979.7 2267.08  4988.0 2264.82  4993.2 2264.44
  4995.5 2262.05  4995.8 2261.55  4999.5 2261.55  4999.7 2262.05  5003.3 2262.05
  5009.9 2263.19  5016.1 2262.28  5030.8 2265.47  5037.5 2272.92  5045.5 2274.96
  5051.6 2274.91  5060.2 2276.85  5066.3 2277.48  5074.6 2279.63  5081.0 2283.83
  5101.9 2291.53  5110.4 2294.15  5116.6 2295.36  5120.9 2297.29  5124.0 2297.29
#Mann=3,-1,0
  4896.7    0.16       0  4995.5    0.07       0  4999.7    0.16       0
Bank Sta=4995.5,4999.7
Exp/Cntr=0.3,0.1

Type RM Length L Ch R = 1,17512,88,88,88
BEGIN DESCRIPTION:
Elm 52 17511.63
END DESCRIPTION:
XS GIS Cut Line= 3
      1510500.90      6765240.11      1510598.13      6765128.99
      1510646.60      6765002.62
#Sta/Elev= 30
  4853.9 2281.28  4894.0 2279.90  4914.9 2277.86  4922.5 2277.84  4936.4 2276.10
  4950.0 2274.13  4957.6 2272.47  4964.2 2272.25  4978.5 2266.26  4986.1 2262.25
  4992.7 2261.63  5004.2 2262.02  5005.3 2260.38  5005.5 2259.88  5009.2 2259.88
  5009.5 2260.38  5013.3 2260.72  5024.0 2262.74  5032.0 2264.62  5037.4 2268.41
  5045.5 2274.74  5056.2 2280.56  5067.4 2290.24  5077.6 2295.48  5086.7 2300.56
  5092.1 2302.58  5109.7 2303.00  5116.8 2304.17  5122.1 2305.36  5136.9 2306.66
#Mann=3,-1,0
  4853.9    0.16       0  5005.3    0.07       0  5009.5    0.16       0
Bank Sta=5005.3,5009.5
Exp/Cntr=0.3,0.1

Type RM Length L Ch R = 1,17424,155,155,155
BEGIN DESCRIPTION:
Elm 52 17423.57
END DESCRIPTION:
XS GIS Cut Line= 3
      1510504.39      6765307.81      1510655.43      6765194.97
      1510747.10      6765082.54
#Sta/Elev= 30
  4814.2 2280.19  4821.7 2279.43  4828.0 2280.11  4857.2 2280.49  4892.6 2279.38
  4907.2 2277.71  4921.8 2274.97  4942.6 2274.67  4951.0 2273.16  4957.2 2274.01
  4964.8 2271.52  4971.8 2267.84  4978.0 2267.84  4992.6 2265.16  4999.4 2262.02
  5002.7 2262.02  5012.0 2257.88  5012.2 2257.38  5016.2 2257.88  5022.0 2257.89
  5028.4 2261.44  5036.4 2263.37  5042.8 2268.44  5057.2 2275.17  5063.6 2284.65
  5071.5 2290.42  5078.0 2297.45  5092.3 2299.14  5121.1 2300.16  5147.8 2302.32
#Mann=3,-1,0
  4814.2    0.16       0  5012.0    0.07       0  5016.2    0.16       0
Bank Sta=5012,5016.2
Exp/Cntr=0.3,0.1

Type RM Length L Ch R = 1,17269,96,96,96
BEGIN DESCRIPTION:
Elm 52 17269.03
END DESCRIPTION:
XS GIS Cut Line= 3
      1510485.27      6765366.84      1510651.95      6765352.95
      1510781.12      6765280.62
#Sta/Elev= 30
  4828.8 2279.39  4848.6 2279.33  4888.7 2277.42  4918.8 2273.44  4928.9 2272.76
  4948.9 2269.96  4979.1 2258.42  4987.0 2255.88  4987.2 2255.38  4990.9 2255.38
  4991.2 2255.88  4994.8 2257.31  5000.7 2257.55  5010.9 2257.16  5016.6 2258.62
  5022.5 2257.51  5032.6 2259.10  5038.3 2258.46  5054.2 2263.54  5060.0 2264.48
  5068.3 2272.28  5075.9 2282.99  5081.7 2281.48  5091.2 2286.94  5103.4 2287.50
  5113.6 2287.41  5119.3 2288.23  5135.3 2287.75  5141.0 2288.45  5144.1 2288.24
#Mann=3,-1,0
  4828.8    0.16       0  4987.0    0.07       0  4991.2    0.16       0
Bank Sta=4987,4991.2
Exp/Cntr=0.3,0.1

Type RM Length L Ch R = 1,17173,135,135,135
BEGIN DESCRIPTION:
Elm 52 17173.379
END DESCRIPTION:
XS GIS Cut Line= 3
      1510555.03      6765438.00      1510655.36      6765446.68
      1510754.97      6765388.02
#Sta/Elev= 30
  4899.3 2276.05  4901.8 2276.05  4909.3 2274.66  4929.4 2270.01  4949.5 2264.69
  4955.9 2262.54  4960.9 2262.51  4969.5 2255.77  4977.5 2254.60  4977.7 2254.10
  4981.4 2254.10  4981.7 2254.60  4989.6 2255.41  4997.3 2257.20  5002.7 2257.20
  5012.1 2259.13  5027.8 2259.23  5034.4 2258.66  5043.4 2262.86  5049.2 2261.79
  5057.6 2266.87  5064.9 2270.65  5070.7 2270.79  5080.6 2274.14  5086.4 2275.47
  5092.4 2278.84  5102.0 2280.56  5107.8 2282.05  5112.7 2282.71  5115.6 2282.71
#Mann=3,-1,0
  4899.3    0.16       0  4977.5    0.07       0  4981.7    0.16       0
Bank Sta=4977.5,4981.7
Exp/Cntr=0.3,0.1

Type RM Length L Ch R = 1,17038,78,78,78
BEGIN DESCRIPTION:
Elm 52 17037.99
END DESCRIPTION:
XS GIS Cut Line= 3
      1510551.25      6765752.27      1510688.41      6765569.97
      1510781.05      6765436.15
#Sta/Elev= 30
  4772.9 2294.48  4778.7 2294.48  4821.4 2290.45  4850.5 2285.78  4856.8 2285.44
  4865.1 2283.58  4871.4 2277.20  4878.4 2273.85  4885.9 2271.84  4892.2 2265.36
  4900.5 2263.87  4906.8 2260.56  4915.1 2260.04  4935.9 2255.91  4942.2 2253.88
  4956.7 2255.05  4976.3 2252.98  4976.6 2252.48  4980.6 2252.98  4985.9 2254.96
  4992.2 2254.98  5006.7 2257.35  5015.5 2260.20  5021.5 2265.55  5036.4 2262.30
  5042.5 2264.90  5051.3 2265.36  5057.4 2267.70  5122.9 2271.87  5163.8 2277.61
#Mann=3,-1,0
  4772.9    0.16       0  4976.3    0.07       0  4980.6    0.16       0
Bank Sta=4976.3,4980.6
Exp/Cntr=0.3,0.1

Type RM Length L Ch R = 1,16960,64,64,64
BEGIN DESCRIPTION:
Elm 52 16959.84
END DESCRIPTION:
XS GIS Cut Line= 3
      1510620.72      6765790.43      1510761.33      6765594.27
      1510844.65      6765455.40
#Sta/Elev= 30
  4761.3 2291.73  4765.9 2291.73  4773.8 2289.67  4776.9 2290.54  4780.0 2291.41
  4788.6 2289.78  4794.7 2290.68  4801.2 2288.66  4809.5 2287.54  4815.6 2287.88
  4824.2 2286.78  4830.3 2284.46  4845.1 2268.71  4851.2 2264.98  4859.8 2262.23
  4887.3 2258.60  4924.2 2257.67  4931.1 2255.79  4960.5 2255.61  4985.4 2250.45
  4985.7 2249.95  4989.7 2250.45  5001.5 2255.58  5010.0 2264.22  5017.7 2268.12
  5023.5 2267.60  5033.2 2268.91  5060.4 2269.38  5134.3 2275.59  5164.6 2276.55
#Mann=4,-1,0
  4761.3    0.07       0  4776.9    0.16       0  4985.4    0.07       0
  4989.7    0.16       0
Bank Sta=4985.4,4989.7
Exp/Cntr=0.3,0.1

Type RM Length L Ch R = 1,16896,89,89,89
BEGIN DESCRIPTION:
Elm 52 16895.61
END DESCRIPTION:
XS GIS Cut Line= 3
      1510728.34      6765807.83      1510808.20      6765641.15
      1510867.02      6765492.38
#Sta/Elev= 30
  4809.0 2294.79  4812.2 2296.06  4819.9 2294.80  4830.7 2294.73  4836.3 2296.14
  4858.9 2293.45  4864.5 2294.40  4875.3 2294.09  4881.6 2291.04  4887.1 2290.76
  4897.5 2281.52  4904.2 2274.28  4909.8 2274.52  4919.7 2267.45  4926.9 2260.82
  4932.4 2260.40  4941.9 2255.77  4964.1 2254.13  4984.1 2250.20  4984.4 2249.70
  4988.4 2250.20  5008.0 2251.87  5025.0 2257.52  5054.7 2255.79  5072.5 2264.68
  5079.1 2269.21  5084.5 2269.20  5094.0 2271.55  5133.2 2273.86  5153.8 2273.99
#Mann=4,-1,0
  4809.0    0.07       0  4812.2    0.16       0  4984.1    0.07       0
  4988.4    0.16       0
Bank Sta=4984.1,4988.4
Exp/Cntr=0.3,0.1

Type RM Length L Ch R = 1,16807,89,89,89
BEGIN DESCRIPTION:
Elm 52 16806.53
END DESCRIPTION:
XS GIS Cut Line= 3
      1510849.88      6765804.31      1510898.48      6765648.09
      1510910.64      6765523.08
#Sta/Elev= 30
  4829.5 2309.05  4857.0 2305.80  4862.9 2299.92  4868.2 2301.50  4888.5 2285.86
  4895.5 2277.82  4900.7 2277.31  4909.4 2270.09  4919.9 2264.40  4928.0 2257.63
  4933.2 2257.15  4940.8 2252.64  4951.3 2251.14  4960.5 2250.99  4970.1 2248.99
  4970.4 2248.49  4974.1 2248.49  4974.4 2248.99  4982.7 2248.99  4990.5 2250.97
  4995.7 2250.97  5003.2 2254.48  5033.4 2253.71  5043.4 2257.16  5063.5 2266.68
  5073.6 2269.36  5083.6 2270.78  5103.7 2271.67  5110.4 2272.71  5118.7 2272.41
#Mann=3,-1,0
  4829.5    0.16       0  4970.1    0.07       0  4974.4    0.16       0
Bank Sta=4970.1,4974.4
Exp/Cntr=0.3,0.1

Type RM Length L Ch R = 1,16718,118,118,118
BEGIN DESCRIPTION:
Elm 52 16718.36
END DESCRIPTION:
XS GIS Cut Line= 3
      1511053.02      6765809.58      1510971.69      6765671.67
      1510955.00      6765538.01
#Sta/Elev= 30
  4839.9 2312.36  4876.6 2311.63  4883.8 2310.52  4889.6 2310.91  4905.2 2308.81
  4911.4 2304.02  4920.9 2293.15  4926.7 2290.11  4934.6 2279.34  4942.3 2273.89
  4948.1 2271.84  4957.8 2266.45  4963.8 2260.52  4969.6 2259.21  4979.4 2254.69
  4985.2 2254.02  4997.1 2247.18  4997.4 2246.68  5001.1 2246.68  5001.4 2247.18
  5004.4 2247.18  5016.2 2248.95  5023.9 2251.46  5033.9 2250.84  5074.2 2251.29
  5084.3 2256.98  5091.9 2263.62  5096.9 2265.62  5104.5 2269.56  5134.7 2271.34
#Mann=3,-1,0
  4839.9    0.16       0  4997.1    0.07       0  5001.4    0.16       0
Bank Sta=4997.1,5001.4
Exp/Cntr=0.3,0.1

Type RM Length L Ch R = 1,16600,204,204,204
BEGIN DESCRIPTION:
Elm 52 16599.97
END DESCRIPTION:
XS GIS Cut Line= 3
      1511131.14      6765714.10      1511058.20      6765592.53
      1511028.84      6765442.25
#Sta/Elev= 30
  4857.0 2304.93  4864.6 2303.65  4874.3 2299.23  4880.1 2293.36  4887.4 2280.46
  4895.7 2271.75  4901.5 2269.11  4910.8 2262.57  4917.1 2256.34  4932.6 2249.14
  4954.0 2249.13  4981.2 2250.26  4990.9 2249.88  4996.8 2249.11  4998.8 2248.16
  5003.6 2248.16  5011.4 2246.06  5011.7 2245.56  5015.4 2245.56  5015.7 2246.06
  5023.8 2247.69  5034.0 2255.63  5040.3 2267.60  5045.4 2268.54  5054.3 2269.09
  5091.8 2269.08  5096.9 2269.80  5125.7 2271.29  5135.8 2270.92  5151.9 2272.01
#Mann=3,-1,0
  4857.0    0.16       0  5011.4    0.07       0  5015.7    0.16       0
Bank Sta=5011.4,5015.7
Exp/Cntr=0.3,0.1

Type RM Length L Ch R = 1,16396,173,173,173
BEGIN DESCRIPTION:
Elm 52 16396.03
END DESCRIPTION:
XS GIS Cut Line= 3
      1511304.72      6765599.47      1511219.66      6765526.56
      1511080.38      6765342.57
#Sta/Elev= 30
  4887.6 2294.02  4910.0 2293.25  4924.2 2281.44  4930.8 2274.58  4952.8 2263.14
  4959.3 2257.16  4966.3 2252.42  4980.2 2244.23  4985.7 2242.32  4986.0 2241.82
  4989.7 2241.82  4990.0 2242.32  4999.4 2243.85  5009.9 2243.52  5016.1 2246.07
  5030.7 2248.05  5037.0 2250.21  5051.5 2251.62  5059.8 2253.48  5066.1 2255.50
  5080.6 2258.47  5086.9 2261.90  5095.2 2261.64  5101.5 2263.95  5116.0 2265.08
  5123.3 2264.81  5186.8 2269.11  5195.1 2268.99  5209.6 2270.80  5230.4 2271.49
#Mann=3,-1,0
  4887.6    0.16       0  4985.7    0.07       0  4990.0    0.16       0
Bank Sta=4985.7,4990
Exp/Cntr=0.3,0.1

Type RM Length L Ch R = 1,16223,165,165,165
BEGIN DESCRIPTION:
Elm 52 16222.829
END DESCRIPTION:
XS GIS Cut Line= 3
      1511404.97      6765487.96      1511340.68      6765402.68
      1511235.31      6765219.30
#Sta/Elev= 30
  4893.2 2287.08  4906.7 2287.27  4921.3 2285.95  4929.6 2278.36  4935.8 2272.06
  4943.2 2268.92  4950.4 2265.24  4971.2 2249.18  4979.5 2244.28  4985.8 2241.28
  4993.3 2240.46  5004.1 2240.12  5004.4 2239.62  5008.2 2239.62  5008.4 2240.12
  5028.5 2246.21  5074.6 2249.08  5081.0 2249.84  5096.8 2253.63  5102.6 2252.89
  5109.2 2256.40  5118.4 2259.40  5124.1 2258.45  5132.3 2260.44  5139.9 2261.34
  5145.7 2260.98  5161.5 2262.05  5177.3 2262.23  5198.9 2264.14  5211.5 2265.89
#Mann=3,-1,0
  4893.2    0.16       0  5004.1    0.07       0  5008.4    0.16       0
Bank Sta=5004.1,5008.4
Exp/Cntr=0.3,0.1

Type RM Length L Ch R = 1,16058,170,170,170
BEGIN DESCRIPTION:
Elm 52 16057.95
END DESCRIPTION:
XS GIS Cut Line= 3
      1511553.00      6765394.62      1511455.77      6765300.87
      1511289.55      6765105.21
#Sta/Elev= 30
  4867.4 2271.42  4898.9 2271.98  4934.2 2271.61  4955.5 2270.61  4962.5 2263.96
  4976.6 2252.66  4983.8 2248.54  4990.8 2242.76  4998.8 2238.25  4999.0 2237.75
  5002.8 2237.75  5003.1 2238.25  5019.3 2239.20  5032.9 2243.28  5054.9 2242.81
  5069.2 2244.18  5083.5 2243.88  5104.3 2244.75  5118.6 2250.12  5132.9 2257.00
  5139.5 2258.68  5153.8 2259.65  5175.8 2259.52  5182.3 2260.12  5196.6 2259.21
  5210.9 2259.23  5217.4 2260.07  5225.2 2259.58  5239.5 2260.62  5259.2 2264.13
#Mann=3,-1,0
  4867.4    0.16       0  4998.8    0.07       0  5003.1    0.16       0
Bank Sta=4998.8,5003.1
Exp/Cntr=0.3,0.1

Type RM Length L Ch R = 1,15888,249,249,249
BEGIN DESCRIPTION:
Elm 52 15887.92
END DESCRIPTION:
XS GIS Cut Line= 2
      1511594.66      6765286.98      1511425.13      6764911.59
#Sta/Elev= 30
  4857.5 2267.40  4870.8 2266.02  4888.5 2259.82  4900.3 2250.28  4917.1 2243.00
  4955.1 2241.30  4963.3 2239.76  4966.6 2236.24  4966.9 2235.74  4970.7 2235.74
  4971.0 2236.24  4986.4 2236.52  4991.9 2237.54  5009.6 2237.44  5015.0 2239.02
  5038.2 2238.21  5043.7 2239.60  5075.8 2241.68  5084.4 2243.83  5089.9 2247.58
  5097.8 2250.48  5119.7 2255.31  5152.6 2257.58  5182.4 2261.74  5211.0 2267.36
  5240.4 2278.30  5251.4 2281.55  5257.2 2284.96  5262.7 2286.18  5269.4 2289.27
#Mann=3,-1,0
  4857.5    0.16       0  4966.6    0.07       0  4971.0    0.16       0
Bank Sta=4966.6,4971
Exp/Cntr=0.3,0.1

Type RM Length L Ch R = 1,15639,133,133,133
BEGIN DESCRIPTION:
Elm 52 15639.18
END DESCRIPTION:
XS GIS Cut Line= 3
      1511601.61      6765266.11      1511639.80      6765007.47
      1511540.83      6764767.85
#Sta/Elev= 30
  4659.6 2265.97  4667.8 2264.55  4677.9 2259.61  4698.1 2247.54  4715.2 2242.73
  4870.0 2239.53  4910.4 2240.33  4931.3 2239.43  4952.9 2239.96  4963.7 2239.56
  4971.0 2238.51  4976.4 2235.91  4985.4 2234.32  4998.2 2233.54  4998.5 2233.04
  5002.6 2233.54  5007.0 2233.66  5017.8 2239.25  5029.7 2254.92  5048.2 2268.57
  5053.6 2270.97  5061.1 2275.74  5071.9 2279.79  5077.5 2283.02  5115.2 2291.59
  5130.8 2293.50  5136.9 2296.39  5147.7 2296.80  5169.3 2301.86  5180.3 2303.04
#Mann=3,-1,0
  4659.6    0.16       0  4998.2    0.07       0  5002.6    0.16       0
Bank Sta=4998.2,5002.6
Exp/Cntr=0.3,0.1

Type RM Length L Ch R = 1,15506,255,255,255
BEGIN DESCRIPTION:
Elm 52 15505.76
END DESCRIPTION:
XS GIS Cut Line= 3
      1511618.97      6765259.20      1511707.51      6764849.48
      1511679.87      6764664.62
#Sta/Elev= 30
  4576.5 2264.51  4582.1 2263.98  4588.0 2261.63  4608.4 2250.21  4626.3 2243.93
  4631.4 2245.17  4639.1 2243.23  4669.8 2241.95  4792.6 2239.87  4802.8 2238.91
  4823.3 2238.32  4884.7 2238.40  4911.5 2239.35  4935.8 2236.45  4960.8 2235.42
  4984.8 2231.63  4985.1 2231.13  4988.9 2231.13  4989.2 2231.63  4993.9 2236.96
  4999.0 2236.96  5007.3 2250.95  5044.6 2278.64  5049.6 2284.33  5068.0 2287.14
  5108.4 2290.79  5128.6 2293.74  5159.0 2295.58  5177.9 2295.66  5182.6 2296.83
#Mann=3,-1,0
  4576.5    0.16       0  4984.8    0.07       0  4989.2    0.16       0
Bank Sta=4984.8,4989.2
Exp/Cntr=0.3,0.1

Type RM Length L Ch R = 1,15251,127,127,127
BEGIN DESCRIPTION:
Elm 52 15250.64
END DESCRIPTION:
XS GIS Cut Line= 3
      1511604.98      6765288.02      1511944.74      6764888.97
      1512055.03      6764837.99
#Sta/Elev= 30
  4475.9 2266.91  4532.5 2261.59  4540.2 2257.53  4546.8 2257.38  4554.5 2251.25
  4561.0 2251.98  4575.3 2246.23  4581.9 2246.87  4589.6 2243.94  4681.8 2244.37
  4731.2 2239.93  4794.9 2237.98  4823.5 2234.19  4852.0 2234.98  4872.9 2231.88
  4901.4 2233.22  4950.9 2231.99  4984.5 2227.19  4984.9 2226.69  4989.8 2227.19
  4993.7 2228.79  4997.4 2236.14  5010.0 2237.93  5015.5 2242.44  5032.9 2244.02
  5038.4 2248.51  5055.4 2250.33  5077.4 2258.97  5089.8 2265.96  5121.5 2278.02
#Mann=3,-1,0
  4475.9    0.16       0  4984.5    0.07       0  4989.8    0.16       0
Bank Sta=4984.5,4989.8
Exp/Cntr=0.3,0.1

Type RM Length L Ch R = 1,15124,211,211,211
BEGIN DESCRIPTION:
Elm 52 15124.29
END DESCRIPTION:
XS GIS Cut Line= 3
      1511690.13      6765278.32      1511936.68      6765000.52
      1512198.86      6764950.17
#Sta/Elev= 30
  4559.4 2257.40  4584.6 2255.95  4633.9 2248.04  4669.1 2245.92  4740.2 2239.00
  4811.2 2236.35  4846.4 2232.10  4874.8 2232.82  4889.0 2231.32  4903.2 2232.11
  4929.2 2230.16  4980.0 2229.93  5007.9 2226.33  5008.3 2225.83  5013.2 2226.33
  5019.7 2234.38  5024.8 2233.91  5030.9 2239.45  5061.5 2245.62  5071.7 2249.74
  5076.8 2248.91  5102.2 2260.27  5112.4 2265.67  5122.6 2273.60  5128.7 2280.34
  5133.8 2278.03  5143.0 2283.98  5153.1 2287.53  5180.7 2293.54  5197.8 2295.09
#Mann=3,-1,0
  4559.4    0.16       0  5007.9    0.07       0  5013.2    0.16       0
Bank Sta=5007.9,5013.2
Exp/Cntr=0.3,0.1

Type RM Length L Ch R = 1,14913,121,121,121
BEGIN DESCRIPTION:
Elm 52 14913.12
END DESCRIPTION:
XS GIS Cut Line= 3
      1511693.63      6765319.96      1511884.59      6765198.44
      1512160.36      6765136.00
#Sta/Elev= 30
  4650.7 2258.64  4703.3 2253.40  4733.8 2249.20  4776.1 2247.94  4806.4 2245.06
  4827.7 2235.59  4833.7 2234.93  4848.9 2227.93  4854.8 2226.81  4870.1 2226.45
  4874.3 2227.66  4887.7 2228.43  4928.7 2229.65  4945.5 2227.96  4959.5 2228.67
  4969.7 2227.83  4986.0 2223.42  4986.4 2222.92  4991.3 2223.42  5010.8 2228.17
  5037.0 2231.67  5051.8 2232.13  5062.0 2237.32  5080.1 2253.57  5085.2 2254.71
  5092.8 2262.54  5113.3 2280.88  5123.3 2288.01  5133.8 2291.11  5159.8 2294.94
#Mann=3,-1,0
  4650.7    0.16       0  4986.0    0.07       0  4991.3    0.16       0
Bank Sta=4986,4991.3
Exp/Cntr=0.3,0.1
