HEC-RAS study Elm 52.prj: Elm 52 Base Level Engineering

--- Elm 52.g01 (geometry) --- (continued)

Type RM Length L Ch R = 1,14792,208,208,208
BEGIN DESCRIPTION:
Elm 52 14791.7
END DESCRIPTION:
XS GIS Cut Line= 3
      1511693.64      6765370.31      1511952.30      6765276.56
      1512148.53      6765189.74
#Sta/Elev= 30
  4725.6 2259.04  4781.0 2255.24  4867.5 2242.95  4886.6 2236.99  4892.8 2230.23
  4898.2 2231.61  4907.9 2223.74  4915.5 2222.24  4915.9 2221.74  4920.8 2222.24
  5004.9 2223.66  5009.3 2226.07  5014.8 2224.07  5025.5 2226.96  5032.6 2231.07
  5038.1 2227.87  5055.9 2235.54  5061.4 2232.06  5079.2 2241.50  5084.7 2236.51
  5091.2 2241.33  5102.1 2243.06  5108.0 2246.07  5113.4 2243.38  5124.0 2247.74
  5131.3 2253.03  5136.7 2251.88  5189.6 2278.83  5211.2 2287.81  5215.3 2287.81
#Mann=3,-1,0
  4725.6    0.16       0  4915.5    0.07       0  4920.8    0.16       0
Bank Sta=4915.5,4920.8
Exp/Cntr=0.3,0.1

Type RM Length L Ch R = 1,14584,134,134,134
BEGIN DESCRIPTION:
Elm 52 14584.49
END DESCRIPTION:
XS GIS Cut Line= 3
      1511761.36      6765545.65      1511928.00      6765462.33
      1512177.44      6765202.49
#Sta/Elev= 30
  4813.1 2255.26  4843.3 2254.60  4888.0 2251.66  4910.3 2249.36  4927.1 2244.20
  4940.2 2243.17  4949.5 2242.77  4962.5 2243.99  4971.8 2238.06  4977.4 2236.21
  4984.9 2225.68  4994.2 2219.45  4996.0 2219.41  4996.4 2218.91  5001.3 2219.41
  5028.7 2224.18  5049.8 2223.12  5071.1 2223.60  5078.1 2226.89  5092.2 2229.26
  5127.7 2231.02  5177.1 2240.83  5226.8 2243.59  5247.9 2248.22  5262.0 2253.34
  5304.5 2272.64  5325.6 2284.36  5332.8 2285.99  5339.7 2289.13  5359.6 2292.81
#Mann=3,-1,0
  4813.1    0.16       0  4996.0    0.07       0  5001.3    0.16       0
Bank Sta=4996,5001.3
Exp/Cntr=0.3,0.1

Type RM Length L Ch R = 1,14450,165,165,165
BEGIN DESCRIPTION:
Elm 52 14449.53
END DESCRIPTION:
XS GIS Cut Line= 3
      1511874.19      6765646.34      1512059.94      6765488.37
      1512190.10      6765264.49
#Sta/Elev= 30
  4763.6 2250.60  4790.9 2249.43  4812.8 2246.63  4841.4 2244.61  4905.1 2241.35
  4911.7 2238.94  4919.4 2239.32  4925.9 2235.99  4933.7 2235.11  4940.2 2231.18
  4947.9 2229.53  4954.5 2223.59  4961.6 2221.44  4975.3 2218.06  4994.7 2217.94
  4995.1 2217.44  5000.0 2217.94  5010.6 2219.75  5026.3 2226.42  5042.1 2226.55
  5063.6 2228.89  5085.1 2237.14  5100.4 2240.65  5158.2 2242.57  5181.1 2244.52
  5202.6 2252.53  5239.2 2272.14  5251.4 2280.51  5261.4 2283.85  5266.4 2286.86
#Mann=3,-1,0
  4763.6    0.16       0  4994.7    0.07       0  5000.0    0.16       0
Bank Sta=4994.7,5000
Exp/Cntr=0.3,0.1

Type RM Length L Ch R = 1,14285,68,68,68
BEGIN DESCRIPTION:
Elm 52 14285.288
END DESCRIPTION:
XS GIS Cut Line= 3
      1511929.77      6765703.63      1512191.81      6765574.34
      1512305.02      6765537.99
#Sta/Elev= 30
  4707.8 2247.35  4731.1 2243.54  4753.5 2242.21  4759.1 2242.62  4776.0 2241.74
  4781.6 2242.33  4791.7 2241.38  4820.9 2240.61  4826.5 2241.44  4880.9 2238.02
  4893.8 2235.98  4903.2 2233.61  4916.3 2228.56  4938.7 2222.96  4947.8 2222.50
  4983.6 2216.99  4992.4 2216.99  4996.3 2216.17  4996.7 2215.67  5001.6 2216.17
  5033.4 2221.08  5038.6 2223.35  5045.4 2228.88  5065.5 2241.61  5087.4 2266.59
  5097.6 2275.05  5102.8 2281.10  5108.4 2285.90  5116.3 2288.20  5118.9 2288.20
#Mann=3,-1,0
  4707.8    0.16       0  4996.3    0.07       0  5001.6    0.16       0
Bank Sta=4996.3,5001.6
Exp/Cntr=0.3,0.1

Type RM Length L Ch R = 1,14217,105,105,105
BEGIN DESCRIPTION:
Elm 52 14217.18
END DESCRIPTION:
XS GIS Cut Line= 3
      1511919.27      6765741.86      1512204.04      6765639.41
      1512355.05      6765609.90
#Sta/Elev= 30
  4696.1 2248.51  4720.2 2245.63  4725.5 2246.60  4750.9 2241.66  4837.7 2237.83
  4843.0 2238.50  4868.4 2234.03  4873.8 2234.66  4924.5 2228.24  4929.9 2228.94
  4936.0 2226.50  4946.6 2225.84  4955.3 2223.74  4960.6 2225.15  4967.9 2221.01
  4978.5 2217.88  4986.0 2215.79  4991.3 2216.80  4993.9 2215.38  4994.3 2214.88
  4999.2 2215.38  5020.1 2215.49  5033.8 2217.76  5050.7 2229.19  5080.2 2255.20
  5085.3 2256.96  5091.4 2264.56  5101.6 2272.25  5122.0 2293.31  5152.6 2296.59
#Mann=3,-1,0
  4696.1    0.16       0  4993.9    0.07       0  4999.2    0.16       0
Bank Sta=4993.9,4999.2
Exp/Cntr=0.3,0.1

Type RM Length L Ch R = 1,14112,69,69,69
BEGIN DESCRIPTION:
Elm 52 14111.89
END DESCRIPTION:
XS GIS Cut Line= 3
      1511938.39      6765764.41      1512164.11      6765731.42
      1512394.98      6765717.54
#Sta/Elev= 30
  4770.6 2247.21  4781.3 2246.33  4807.6 2241.75  4851.3 2238.57  4888.4 2232.92
  4916.2 2230.27  4959.2 2228.26  4969.3 2226.81  4991.2 2221.92  4996.6 2217.34
  5001.7 2217.34  5007.0 2212.83  5007.4 2212.33  5012.3 2212.83  5019.6 2213.94
  5049.7 2215.18  5059.7 2214.80  5069.7 2213.11  5079.8 2214.69  5089.8 2218.40
  5099.8 2225.18  5119.8 2246.65  5129.8 2254.77  5136.9 2268.32  5141.9 2267.26
  5149.9 2280.35  5159.9 2293.50  5169.9 2297.78  5200.0 2303.27  5230.0 2306.96
#Mann=3,-1,0
  4770.6    0.16       0  5007.0    0.07       0  5012.3    0.16       0
Bank Sta=5007,5012.3
Exp/Cntr=0.3,0.1

Type RM Length L Ch R = 1,14043,113,113,113
BEGIN DESCRIPTION:
Elm 52 14042.65
END DESCRIPTION:
XS GIS Cut Line= 3
      1511945.33      6765804.34      1512197.09      6765788.72
      1512349.83      6765786.98
#Sta/Elev= 30
  4749.5 2245.15  4759.2 2244.47  4767.7 2242.57  4772.7 2243.82  4789.2 2239.85
  4819.3 2238.40  4849.4 2235.88  4879.4 2228.47  4889.4 2226.90  4928.5 2223.32
  4933.6 2224.75  4977.0 2212.01  4977.4 2211.51  4982.3 2212.01  4998.2 2214.15
  5009.7 2214.16  5019.7 2215.22  5029.7 2214.41  5039.7 2216.07  5049.7 2222.08
  5059.7 2231.27  5069.7 2242.70  5079.7 2255.30  5089.7 2264.05  5109.7 2284.93
  5119.7 2293.51  5129.7 2295.59  5139.7 2296.28  5149.6 2299.25  5154.5 2299.25
#Mann=3,-1,0
  4749.5    0.16       0  4977.0    0.07       0  4982.3    0.16       0
Bank Sta=4977,4982.3
Exp/Cntr=0.3,0.1

Type RM Length L Ch R = 1,13930,109,109,109
BEGIN DESCRIPTION:
Elm 52 13930.28
END DESCRIPTION:
XS GIS Cut Line= 3
      1511922.77      6765839.06      1512148.48      6765887.67
      1512327.29      6765866.84
#Sta/Elev= 30
  4768.1 2246.73  4801.1 2243.19  4842.0 2237.06  4872.7 2234.58  4903.4 2229.23
  4923.8 2224.50  4934.2 2221.00  4954.5 2218.68  4964.7 2218.45  4978.4 2215.49
  4985.2 2211.99  5002.9 2211.21  5003.3 2210.71  5007.8 2210.71  5008.2 2211.21
  5015.6 2213.82  5025.7 2213.72  5035.0 2216.11  5040.1 2214.72  5045.8 2218.72
  5076.0 2236.62  5096.2 2249.76  5106.2 2257.78  5116.3 2266.99  5123.6 2277.54
  5128.6 2277.03  5136.4 2284.18  5146.5 2287.05  5175.3 2292.40  5179.0 2292.40
#Mann=3,-1,0
  4768.1    0.16       0  5002.9    0.07       0  5008.2    0.16       0
Bank Sta=5002.9,5008.2
Exp/Cntr=0.3,0.1

Type RM Length L Ch R = 1,13821,112,112,112
BEGIN DESCRIPTION:
Elm 52 13821.371
END DESCRIPTION:
XS GIS Cut Line= 3
      1511891.49      6765882.44      1512102.50      6765981.96
      1512254.99      6765938.00
#Sta/Elev= 30
  4766.7 2245.13  4772.1 2244.04  4812.1 2242.04  4848.0 2236.44  4857.6 2236.23
  4880.4 2232.54  4885.9 2230.86  4903.2 2231.12  4925.4 2224.85  4937.0 2220.22
  4969.6 2213.43  4982.6 2213.40  4995.9 2209.51  4996.4 2209.01  5001.3 2209.51
  5013.0 2211.19  5035.7 2211.32  5054.6 2212.70  5064.2 2220.19  5069.4 2217.30
  5075.5 2223.60  5096.3 2236.67  5103.0 2243.41  5108.2 2242.10  5117.1 2248.79
  5136.7 2261.57  5141.9 2259.67  5148.3 2264.74  5156.1 2269.12  5158.7 2269.12
#Mann=3,-1,0
  4766.7    0.16       0  4995.9    0.07       0  5001.3    0.16       0
Bank Sta=4995.9,5001.3
Exp/Cntr=0.3,0.1

Type RM Length L Ch R = 1,13709,153,153,153
BEGIN DESCRIPTION:
Elm 52 13708.76
END DESCRIPTION:
XS GIS Cut Line= 3
      1511803.02      6765974.49      1512023.48      6766064.76
      1512285.65      6766063.02
#Sta/Elev= 30
  4758.1 2245.34  4807.9 2242.62  4825.1 2243.07  4837.3 2242.00  4890.7 2233.42
  4909.3 2231.34  4914.7 2229.93  4922.3 2228.97  4933.1 2228.30  4938.7 2227.18
  4954.7 2223.14  4962.7 2220.21  4976.4 2213.96  4986.7 2211.55  5017.8 2210.92
  5045.1 2208.87  5045.6 2208.37  5050.1 2208.37  5050.5 2208.87  5067.8 2215.42
  5087.8 2219.89  5097.8 2222.96  5137.8 2242.00  5147.8 2245.20  5167.8 2247.34
  5187.8 2248.26  5217.9 2251.35  5237.9 2254.62  5255.7 2259.01  5258.5 2259.01
#Mann=3,-1,0
  4758.1    0.16       0  5045.1    0.07       0  5050.5    0.16       0
Bank Sta=5045.1,5050.5
Exp/Cntr=0.3,0.1

Type RM Length L Ch R = 1,13556,124,124,124
BEGIN DESCRIPTION:
Elm 52 13556.47
END DESCRIPTION:
XS GIS Cut Line= 3
      1511730.12      6766155.04      1511955.77      6766189.76
      1512231.73      6766156.99
#Sta/Elev= 30
  4772.0 2253.57  4777.0 2253.57  4823.4 2244.71  4868.0 2241.45  4886.6 2237.96
  4891.7 2238.20  4908.5 2232.53  4948.9 2225.59  4954.9 2223.57  4960.0 2224.12
  4979.3 2220.13  4989.4 2219.50  4997.4 2210.15  5002.4 2210.15  5006.9 2206.63
  5007.3 2206.13  5012.3 2206.63  5049.9 2211.38  5080.1 2209.99  5110.3 2211.31
  5120.4 2212.76  5130.4 2218.34  5138.9 2224.98  5144.0 2224.85  5150.6 2230.16
  5170.7 2237.90  5180.8 2240.66  5190.9 2242.34  5221.1 2244.47  5278.2 2245.75
#Mann=3,-1,0
  4772.0    0.16       0  5006.9    0.07       0  5012.3    0.16       0
Bank Sta=5006.9,5012.3
Exp/Cntr=0.3,0.1

Type RM Length L Ch R = 1,13432,167,167,167
BEGIN DESCRIPTION:
Elm 52 13432.3
END DESCRIPTION:
XS GIS Cut Line= 3
      1511669.28      6766373.79      1511976.61      6766307.81
      1512247.47      6766215.79
#Sta/Elev= 30
  4687.6 2273.89  4695.0 2269.66  4734.1 2267.13  4739.2 2263.96  4754.8 2263.20
  4775.3 2259.73  4795.7 2252.76  4838.0 2242.40  4857.1 2239.15  4882.3 2237.66
  4898.0 2232.48  4908.2 2227.37  4926.6 2215.20  4931.7 2217.57  4938.9 2213.35
  4949.1 2211.47  4981.1 2211.07  4995.8 2206.11  4996.2 2205.61  5001.2 2206.11
  5031.9 2208.46  5105.4 2207.62  5148.1 2224.72  5168.1 2226.22  5173.4 2228.54
  5199.5 2232.71  5211.5 2237.31  5230.9 2239.51  5236.2 2241.75  5288.0 2244.49
#Mann=3,-1,0
  4687.6    0.16       0  4995.8    0.07       0  5001.2    0.16       0
Bank Sta=4995.8,5001.2
Exp/Cntr=0.3,0.1

Type RM Length L Ch R = 1,13265,136,136,136
BEGIN DESCRIPTION:
Elm 52 13265.39
END DESCRIPTION:
XS GIS Cut Line= 3
      1511707.49      6766490.11      1512053.00      6766441.49
      1512245.74      6766314.73
#Sta/Elev= 30
  4656.3 2289.70  4694.2 2283.45  4714.4 2276.75  4744.7 2268.67  4774.5 2256.92
  4779.5 2254.79  4785.1 2250.51  4805.3 2243.26  4815.4 2237.34  4845.7 2214.18
  4850.8 2207.56  4865.9 2205.94  4966.8 2205.89  4998.3 2204.08  5001.0 2202.76
  5001.4 2202.26  5006.4 2202.76  5023.1 2203.93  5031.5 2206.89  5038.2 2210.95
  5044.2 2210.55  5053.3 2212.32  5103.4 2213.43  5131.6 2217.19  5161.7 2228.24
  5167.7 2229.49  5182.8 2236.26  5197.9 2239.90  5211.1 2241.51  5235.9 2241.75
#Mann=3,-1,0
  4656.3    0.16       0  5001.0    0.07       0  5006.4    0.16       0
Bank Sta=5001,5006.4
Exp/Cntr=0.3,0.1

Type RM Length L Ch R = 1,13129,120,120,120
BEGIN DESCRIPTION:
Elm 52 13129.07
END DESCRIPTION:
XS GIS Cut Line= 3
      1511782.15      6766668.93      1512007.86      6766563.02
      1512235.31      6766356.41
#Sta/Elev= 30
  4752.9 2289.62  4774.8 2287.55  4815.4 2282.66  4822.3 2279.50  4855.5 2270.78
  4861.0 2267.95  4877.6 2263.27  4883.8 2259.37  4929.5 2240.19  4952.3 2232.18
  4957.8 2228.62  4975.1 2220.96  4980.6 2216.80  4988.0 2208.97  4997.9 2203.17
  5015.2 2201.64  5015.6 2201.14  5020.6 2201.64  5032.1 2202.65  5046.3 2206.47
  5053.0 2207.09  5088.8 2206.43  5109.8 2209.97  5180.7 2212.44  5209.1 2212.22
  5223.3 2213.56  5244.2 2221.10  5280.1 2236.16  5301.0 2240.86  5309.5 2241.33
#Mann=4,-1,0
  4752.9    0.07       0  4774.8    0.16       0  5015.2    0.07       0
  5020.6    0.16       0
Bank Sta=5015.2,5020.6
Exp/Cntr=0.3,0.1

Type RM Length L Ch R = 1,13009,85,85,85
BEGIN DESCRIPTION:
Elm 52 13009.3
END DESCRIPTION:
XS GIS Cut Line= 3
      1511855.09      6766783.50      1512106.82      6766590.80
      1512257.88      6766378.96
#Sta/Elev= 30
  4679.3 2274.01  4694.0 2273.22  4747.2 2269.89  4776.2 2257.09  4797.1 2254.39
  4805.1 2251.12  4811.6 2246.91  4817.9 2246.06  4826.1 2241.18  4855.1 2231.75
  4861.4 2231.52  4868.1 2228.49  4890.5 2222.10  4905.0 2219.15  4911.3 2219.05
  4954.9 2203.71  4987.5 2200.45  4987.9 2199.95  4992.9 2200.45  5003.8 2200.48
  5018.6 2204.08  5054.2 2205.56  5061.2 2208.56  5069.0 2209.74  5155.0 2211.65
  5169.8 2215.12  5196.8 2227.74  5226.3 2238.50  5233.1 2240.37  5256.5 2240.10
#Mann=4,-1,0
  4679.3    0.07       0  4694.0    0.16       0  4987.5    0.07       0
  4992.9    0.16       0
Bank Sta=4987.5,4992.9
Exp/Cntr=0.3,0.1

Type RM Length L Ch R = 1,12924,126,126,126
BEGIN DESCRIPTION:
Elm 52 12924.13
END DESCRIPTION:
XS GIS Cut Line= 3
      1511952.31      6766849.47      1512186.68      6766615.10
      1512322.09      6766352.96
#Sta/Elev= 30
  4671.3 2263.93  4681.3 2262.52  4716.7 2247.21  4745.0 2238.01  4759.1 2234.71
  4773.2 2232.32  4808.6 2229.43  4851.0 2219.38  4865.2 2218.36  4879.3 2215.02
  4900.5 2212.36  4921.7 2206.38  4950.0 2201.35  4978.3 2201.71  5002.7 2200.25
  5010.5 2198.58  5010.9 2198.08  5015.9 2198.58  5029.7 2200.75  5051.8 2208.22
  5112.0 2209.33  5134.5 2211.25  5162.6 2218.78  5168.3 2223.61  5184.7 2229.17
  5190.8 2232.97  5201.3 2235.74  5213.3 2236.99  5229.0 2236.15  5297.8 2241.39
#Mann=3,-1,0
  4671.3    0.16       0  5010.5    0.07       0  5015.9    0.16       0
Bank Sta=5010.5,5015.9
Exp/Cntr=0.3,0.1

Type RM Length L Ch R = 1,12798,91,91,91
BEGIN DESCRIPTION:
Elm 52 12797.54
END DESCRIPTION:
XS GIS Cut Line= 3
      1512040.86      6766840.79      1512282.16      6766701.91
      1512537.34      6766469.30
#Sta/Elev= 30
  4730.5 2235.50  4770.9 2229.59  4820.2 2225.58  4829.8 2223.72  4845.6 2223.01
  4851.4 2220.73  4941.9 2207.27  4969.2 2201.00  4977.6 2201.00  4985.0 2198.49
  5006.2 2197.08  5006.6 2196.58  5011.6 2197.08  5020.8 2197.19  5041.8 2206.58
  5049.2 2205.85  5098.5 2208.62  5155.3 2209.46  5183.7 2212.46  5226.2 2220.42
  5233.0 2223.16  5240.4 2223.31  5247.2 2226.04  5254.6 2226.15  5268.8 2228.93
  5275.5 2232.16  5283.0 2233.21  5318.1 2244.02  5346.5 2250.80  5354.2 2250.91
#Mann=4,-1,0
  4730.5    0.07       0  4820.2    0.16       0  5006.2    0.07       0
  5011.6    0.16       0
Bank Sta=5006.2,5011.6
Exp/Cntr=0.3,0.1

Type RM Length L Ch R = 1,12707,98,98,98
BEGIN DESCRIPTION:
Elm 52 12706.79
END DESCRIPTION:
XS GIS Cut Line= 3
      1512079.00      6766894.63      1512337.72      6766771.35
      1512605.94      6766522.16
#Sta/Elev= 30
  4712.0 2238.64  4714.5 2235.16  4720.0 2233.35  4737.2 2230.89  4765.4 2230.60
  4788.1 2235.44  4810.8 2233.24  4843.1 2221.46  4884.8 2211.34  4929.8 2207.68
  4952.5 2199.44  5003.5 2195.86  5003.9 2195.36  5009.1 2195.86  5048.8 2203.59
  5197.3 2205.68  5204.2 2208.51  5211.5 2208.57  5218.3 2212.96  5225.7 2212.87
  5232.5 2217.26  5239.8 2217.10  5246.7 2221.16  5254.0 2220.95  5260.8 2225.19
  5275.0 2227.41  5289.2 2232.54  5296.0 2237.77  5317.5 2245.81  5364.7 2254.14
#Mann=4,-1,0
  4712.0    0.07       0  4843.1    0.16       0  5003.5    0.07       0
  5009.1    0.16       0
Bank Sta=5003.5,5009.1
Exp/Cntr=0.3,0.1

Type RM Length L Ch R = 1,12609,141,141,141
BEGIN DESCRIPTION:
Elm 52 12609.49
END DESCRIPTION:
XS GIS Cut Line= 3
      1512110.30      6767016.14      1512405.43      6766840.80
      1512664.14      6766554.30
#Sta/Elev= 30
  4649.7 2233.45  4658.4 2235.40  4674.0 2230.56  4711.0 2233.63  4716.9 2231.15
  4783.2 2225.12  4812.3 2217.74  4833.7 2216.17  4849.4 2213.47  4855.2 2213.92
  4870.8 2210.82  4987.7 2203.30  4990.8 2200.57  5001.6 2199.73  5013.0 2193.43
  5013.5 2192.93  5018.6 2193.43  5051.0 2196.94  5058.4 2199.68  5086.8 2203.26
  5192.9 2202.68  5228.1 2205.04  5270.7 2211.11  5284.9 2218.10  5306.5 2231.65
  5313.3 2234.50  5327.5 2244.69  5334.2 2246.58  5341.7 2250.64  5379.0 2257.30
#Mann=4,-1,0
  4649.7    0.07       0  4783.2    0.16       0  5013.0    0.07       0
  5018.6    0.16       0
Bank Sta=5013,5018.6
Exp/Cntr=0.3,0.1

Type RM Length L Ch R = 1,12468,110,110,110
BEGIN DESCRIPTION:
Elm 52 12467.94
END DESCRIPTION:
XS GIS Cut Line= 3
      1512315.16      6767165.44      1512546.05      6766846.01
      1512772.25      6766631.90
#Sta/Elev= 30
  4598.8 2235.17  4625.3 2232.79  4646.2 2228.33  4675.6 2216.88  4690.3 2207.64
  4711.2 2203.43  4719.0 2197.27  4725.9 2195.83  4776.2 2202.74  4832.6 2200.57
  4912.3 2201.64  4941.1 2200.46  4962.6 2195.56  4995.0 2192.22  4995.5 2191.72
  5000.6 2192.22  5012.0 2195.85  5019.0 2200.19  5026.2 2201.18  5089.7 2202.44
  5118.0 2204.81  5188.8 2215.40  5202.9 2222.43  5238.5 2245.78  5252.7 2252.34
  5280.7 2260.02  5287.9 2259.48  5294.8 2262.43  5302.1 2262.56  5304.4 2265.11
#Mann=3,-1,0
  4598.8    0.16       0  4995.0    0.07       0  5000.6    0.16       0
Bank Sta=4995,5000.6
Exp/Cntr=0.3,0.1

Type RM Length L Ch R = 1,12358,149,149,149
BEGIN DESCRIPTION:
Elm 52 12358.09
END DESCRIPTION:
XS GIS Cut Line= 3
      1512304.97      6767238.03      1512632.16      6766914.41
      1512855.02      6766938.00
#Sta/Elev= 30
  4539.8 2241.80  4561.1 2240.48  4624.7 2229.80  4631.8 2225.37  4638.8 2225.11
  4645.9 2219.84  4652.9 2218.72  4660.1 2213.33  4667.1 2212.21  4688.3 2202.31
  4737.8 2201.53  4751.9 2195.49  4759.1 2194.90  4773.2 2200.13  4893.4 2200.66
  4949.9 2197.13  4975.4 2190.05  4975.9 2189.55  4981.0 2190.05  4992.4 2192.77
  5012.9 2193.43  5053.1 2210.53  5103.4 2217.33  5123.5 2223.06  5153.7 2236.28
  5172.7 2248.03  5177.7 2248.65  5183.9 2254.11  5214.0 2271.52  5224.1 2274.91
#Mann=3,-1,0
  4539.8    0.16       0  4975.4    0.07       0  4981.0    0.16       0
Bank Sta=4975.4,4981
Exp/Cntr=0.3,0.1

Type RM Length L Ch R = 1,12209,104,104,104
BEGIN DESCRIPTION:
Elm 52 12209.18
END DESCRIPTION:
XS GIS Cut Line= 3
      1512332.55      6767238.34      1512651.95      6767057.81
      1512867.23      6766964.06
#Sta/Elev= 30
  4629.3 2240.07  4660.7 2233.62  4682.3 2225.29  4698.2 2216.01  4704.0 2215.66
  4719.9 2205.24  4725.6 2205.41  4741.5 2199.95  4792.9 2197.73  4806.5 2190.67
  4828.1 2197.76  4865.7 2198.05  4946.5 2196.57  5018.5 2189.65  5019.0 2189.15
  5024.1 2189.65  5030.0 2193.25  5035.5 2193.08  5043.1 2202.39  5053.5 2209.12
  5075.9 2211.69  5111.2 2220.75  5129.2 2229.41  5134.7 2230.03  5152.2 2241.04
  5158.1 2246.76  5187.0 2257.51  5205.0 2269.06  5217.7 2274.73  5231.0 2276.03
#Mann=3,-1,0
  4629.3    0.16       0  5018.5    0.07       0  5024.1    0.16       0
Bank Sta=5018.5,5024.1
Exp/Cntr=0.3,0.1

Type RM Length L Ch R = 1,12105,119,119,119
BEGIN DESCRIPTION:
Elm 52 12104.86
END DESCRIPTION:
XS GIS Cut Line= 3
      1512342.93      6767250.52      1512650.22      6767163.72
      1512868.49      6767002.61
#Sta/Elev= 30
  4675.4 2238.11  4703.3 2233.53  4737.3 2213.79  4742.5 2213.08  4750.3 2207.31
  4771.1 2198.23  4849.6 2195.62  4872.2 2187.77  4872.6 2187.27  4877.8 2187.77
  4895.8 2194.41  4928.0 2195.08  4968.5 2189.45  5001.4 2189.39  5024.4 2194.22
  5030.7 2193.04  5045.3 2199.49  5051.5 2199.20  5074.6 2206.35  5130.9 2213.96
  5166.4 2225.61  5181.0 2238.89  5187.2 2239.86  5195.6 2246.59  5201.9 2247.55
  5210.3 2253.67  5216.5 2253.50  5231.1 2264.52  5245.8 2271.86  5266.0 2275.39
#Mann=3,-1,0
  4675.4    0.16       0  4872.2    0.07       0  4877.8    0.16       0
Bank Sta=4872.2,4877.8
Exp/Cntr=0.3,0.1

Type RM Length L Ch R = 1,11986,239,239,239
BEGIN DESCRIPTION:
Elm 52 11985.94
END DESCRIPTION:
XS GIS Cut Line= 3
      1512316.91      6767281.77      1512634.59      6767262.67
      1512850.77      6767044.77
#Sta/Elev= 30
  4710.6 2241.10  4715.2 2240.44  4728.7 2238.19  4818.9 2200.58  4919.1 2192.18
  4939.1 2192.20  4959.1 2187.52  4976.4 2187.01  4976.8 2186.51  4982.0 2187.01
  5023.8 2189.74  5032.7 2191.06  5039.5 2194.10  5046.6 2192.45  5053.6 2194.84
  5060.7 2194.22  5067.8 2197.78  5074.9 2196.99  5081.9 2199.95  5089.0 2198.65
  5124.4 2204.35  5131.5 2203.79  5138.5 2205.70  5230.5 2214.25  5258.7 2223.53
  5308.2 2254.18  5315.3 2256.21  5322.4 2261.07  5329.5 2262.57  5335.8 2267.35
#Mann=4,-1,0
  4710.6    0.07       0  4715.2    0.16       0  4976.4    0.07       0
  4982.0    0.16       0
Bank Sta=4976.4,4982
Exp/Cntr=0.3,0.1

Type RM Length L Ch R = 1,11747,112,112,112
BEGIN DESCRIPTION:
Elm 52 11746.83
END DESCRIPTION:
XS GIS Cut Line= 3
      1512212.72      6767467.53      1512526.95      6767439.76
      1512863.74      6767068.25
#Sta/Elev= 30
  4755.3 2247.87  4846.1 2244.22  4878.1 2242.41  4908.2 2238.93  4921.8 2219.95
  4928.2 2207.95  4948.3 2195.05  4958.4 2189.93  4968.4 2186.85  4985.5 2185.23
  4986.0 2184.73  4991.4 2185.23  5028.6 2190.02  5091.8 2191.00  5127.1 2194.54
  5212.1 2194.86  5297.2 2198.84  5445.9 2211.56  5474.3 2216.08  5502.7 2224.78
  5509.4 2228.43  5516.9 2233.84  5523.6 2240.15  5531.1 2243.42  5537.8 2249.33
  5545.3 2253.74  5552.0 2259.55  5566.2 2264.69  5569.4 2270.23  5572.2 2270.23
#Mann=4,-1,0
  4755.3    0.07       0  4846.1    0.16       0  4985.5    0.07       0
  4991.4    0.16       0
Bank Sta=4985.5,4991.4
Exp/Cntr=0.3,0.1

Type RM Length L Ch R = 1,11635,210,210,210
BEGIN DESCRIPTION:
Elm 52 11635.04
END DESCRIPTION:
XS GIS Cut Line= 3
      1512355.07      6767719.28      1512499.18      6767543.92
      1512890.77      6767145.40
#Sta/Elev= 30
  4760.3 2243.16  4839.3 2241.03  4860.8 2238.29  4881.6 2232.27  4888.9 2232.22
  4896.0 2228.55  4903.8 2229.03  4910.3 2224.34  4924.7 2224.29  4931.1 2220.17
  4939.0 2220.15  4959.8 2210.93  4967.7 2199.23  4974.2 2200.88  4981.4 2192.55
  4987.3 2193.90  5002.7 2182.46  5006.7 2182.16  5007.2 2181.66  5012.6 2182.16
  5030.9 2185.97  5087.5 2189.08  5115.8 2188.57  5165.2 2193.14  5250.1 2194.62
  5448.1 2211.36  5469.4 2214.22  5504.7 2223.94  5533.0 2237.49  5546.0 2246.55
#Mann=5,-1,0
  4760.3    0.16       0  4839.3    0.07       0  4888.9    0.16       0
  5006.7    0.07       0  5012.6    0.16       0
Bank Sta=5006.7,5012.6
Exp/Cntr=0.3,0.1

Type RM Length L Ch R = 1,11425,130,130,130
BEGIN DESCRIPTION:
Elm 52 11425.156
END DESCRIPTION:
XS GIS Cut Line= 3
      1512450.58      6767766.14      1512703.22      6767581.70
      1512954.98      6767188.02
#Sta/Elev= 30
  4687.2 2238.61  4717.4 2237.26  4723.6 2235.25  4754.4 2220.23  4781.4 2205.23
  4810.8 2196.65  4840.1 2193.03  4861.0 2196.99  4890.3 2191.50  4932.0 2190.49
  4952.9 2187.75  4989.8 2188.08  5000.0 2185.16  5005.2 2185.16  5017.4 2179.09
  5029.7 2178.41  5030.2 2177.91  5035.6 2178.41  5063.0 2186.01  5069.0 2189.45
  5075.6 2190.99  5193.3 2194.40  5265.5 2200.40  5336.8 2210.39  5387.0 2215.56
  5431.7 2222.40  5453.8 2229.50  5459.7 2229.40  5464.4 2234.17  5467.3 2234.17
#Mann=3,-1,0
  4687.2    0.16       0  5029.7    0.07       0  5035.6    0.16       0
Bank Sta=5029.7,5035.6
Exp/Cntr=0.3,0.1

Type RM Length L Ch R = 1,11295,109,109,109
BEGIN DESCRIPTION:
Elm 52 11294.72
END DESCRIPTION:
XS GIS Cut Line= 3
      1512575.55      6767814.77      1512752.65      6767682.81
      1513050.62      6767194.27
#Sta/Elev= 30
  4769.8 2229.66  4774.1 2226.50  4788.7 2224.15  4794.9 2219.16  4803.3 2215.95
  4824.1 2203.70  4844.9 2193.00  4853.3 2190.72  4888.8 2188.77  4968.0 2188.60
  4981.1 2183.84  4988.9 2176.81  5000.5 2174.34  5001.0 2173.84  5006.4 2174.34
  5040.2 2181.31  5046.1 2184.97  5061.6 2186.25  5067.4 2189.60  5156.4 2191.13
  5251.3 2195.07  5257.1 2197.14  5288.1 2199.32  5309.4 2203.89  5352.0 2205.81
  5388.8 2210.40  5468.2 2213.35  5483.6 2216.47  5526.3 2221.24  5562.9 2230.65
#Mann=3,-1,0
  4769.8    0.16       0  5000.5    0.07       0  5006.4    0.16       0
Bank Sta=5000.5,5006.4
Exp/Cntr=0.3,0.1

Type RM Length L Ch R = 1,11186,89,89,89
BEGIN DESCRIPTION:
Elm 52 11185.87
END DESCRIPTION:
XS GIS Cut Line= 3
      1512683.18      6767859.92      1512860.29      6767693.23
      1513080.41      6767318.85
#Sta/Elev= 30
  4758.9 2226.05  4763.6 2226.05  4768.6 2220.54  4789.7 2207.54  4797.0 2204.54
  4803.8 2199.52  4820.5 2192.49  4832.1 2189.11  4895.2 2187.96  4924.4 2188.35
  4938.6 2183.91  4945.4 2180.42  4973.8 2177.11  4981.1 2177.36  4998.9 2174.08
  4999.4 2173.58  5004.9 2174.08  5008.2 2178.34  5017.6 2186.53  5023.4 2185.40
  5039.1 2188.98  5076.2 2190.72  5082.0 2189.88  5170.6 2194.53  5236.3 2200.65
  5242.1 2199.84  5279.3 2203.63  5396.5 2211.03  5417.9 2214.27  5436.4 2214.20
#Mann=5,-1,0
  4758.9    0.16       0  4820.5    0.07       0  4895.2    0.16       0
  4998.9    0.07       0  5004.9    0.16       0
Bank Sta=4998.9,5004.9
Exp/Cntr=0.3,0.1

Type RM Length L Ch R = 1,11097,123,123,123
BEGIN DESCRIPTION:
Elm 52 11096.59
END DESCRIPTION:
XS GIS Cut Line= 3
      1512757.87      6767905.02      1512922.79      6767757.47
      1513099.39      6767341.93
#Sta/Elev= 30
  4777.3 2215.70  4780.2 2212.20  4787.0 2212.13  4837.3 2193.10  4851.3 2188.70
  4907.6 2187.01  4914.8 2185.93  4929.0 2180.72  4943.2 2178.17  4979.8 2178.23
  5018.1 2173.55  5018.6 2173.05  5024.1 2173.55  5030.6 2173.57  5044.7 2186.23
  5052.3 2187.53  5097.5 2187.20  5144.8 2191.34  5173.9 2191.56  5237.1 2195.78
  5258.8 2197.62  5280.5 2201.94  5303.0 2203.22  5379.3 2212.26  5397.6 2213.11
  5403.0 2214.96  5421.2 2215.83  5426.6 2218.53  5432.6 2219.63  5450.1 2221.05
#Mann=5,-1,0
  4777.3    0.16       0  4837.3    0.07       0  4979.8    0.16       0
  5018.1    0.07       0  5024.1    0.16       0
Bank Sta=5018.1,5024.1
Exp/Cntr=0.3,0.1

Type RM Length L Ch R = 1,10974,260,260,260
BEGIN DESCRIPTION:
Elm 52 10973.66
END DESCRIPTION:
XS GIS Cut Line= 3
      1513002.65      6767917.19      1513033.90      6767793.92
      1513118.97      6767356.39
#Sta/Elev= 30
  4866.0 2196.58  4913.8 2195.74  4955.3 2195.00  4968.3 2193.35  4975.4 2187.47
  4980.6 2190.20  4988.5 2185.40  4993.2 2185.40  4999.2 2178.19  5009.4 2171.92
  5014.0 2171.32  5016.6 2170.98  5017.1 2170.48  5022.6 2170.98  5024.9 2172.86
  5030.0 2171.76  5050.1 2175.44  5070.5 2184.25  5111.3 2184.78  5121.5 2182.57
  5128.2 2183.58  5133.3 2180.86  5179.9 2188.45  5185.0 2186.11  5231.6 2192.13
  5236.7 2190.81  5283.2 2201.07  5315.0 2204.12  5396.7 2219.75  5438.9 2223.33
#Mann=6,-1,0
  4866.0    0.07       0  4913.8    0.16       0  4955.3    0.07       0
  5014.0    0.16       0  5016.6    0.07       0  5022.6    0.16       0
Bank Sta=5016.6,5022.6
Exp/Cntr=0.3,0.1

Type RM Length L Ch R = 1,10714,142,142,142
BEGIN DESCRIPTION:
Elm 52 10714.11
END DESCRIPTION:
XS GIS Cut Line= 3
      1513125.90      6767884.25      1513164.11      6767663.72
      1513160.65      6767421.86
#Sta/Elev= 30
  4710.7 2189.38  4727.2 2188.45  4738.6 2186.24  4747.5 2185.48  4788.1 2186.04
  4793.2 2186.93  4820.1 2187.80  4859.1 2189.18  4879.4 2188.33  4889.6 2187.26
  4899.7 2184.97  4907.6 2182.05  4912.7 2183.53  4919.1 2180.11  4929.8 2176.01
  4934.5 2176.01  4940.2 2172.90  4960.2 2169.89  4970.2 2170.70  4987.2 2168.39
  4987.7 2167.89  4993.2 2168.39  5000.2 2172.38  5010.2 2176.80  5040.2 2198.89
  5050.2 2205.24  5060.2 2209.61  5090.2 2218.19  5140.3 2228.30  5176.4 2236.84
#Mann=5,-1,0
  4710.7    0.16       0  4820.1    0.07       0  4919.1    0.16       0
  4987.2    0.07       0  4993.2    0.16       0
Bank Sta=4987.2,4993.2
Exp/Cntr=0.3,0.1

Type RM Length L Ch R = 1,10572,125,125,125
BEGIN DESCRIPTION:
Elm 52 10572.35
END DESCRIPTION:
XS GIS Cut Line= 3
      1513129.37      6767885.96      1513264.80      6767696.70
      1513408.89      6767458.87
#Sta/Elev= 30
  4768.0 2189.38  4820.7 2182.90  4841.6 2183.49  4871.1 2186.69  4900.6 2184.90
  4906.7 2183.49  4921.5 2185.19  4931.9 2183.84  4942.4 2182.19  4963.3 2181.83
  4992.7 2169.18  4993.9 2164.65  4994.4 2164.15  4999.9 2164.65  5044.7 2171.58
  5066.1 2182.38  5071.9 2186.58  5081.1 2190.42  5087.4 2195.18  5102.9 2202.43
  5124.3 2216.97  5139.5 2225.12  5145.6 2230.53  5166.9 2241.86  5203.8 2271.35
  5209.7 2278.57  5219.3 2285.71  5240.6 2288.19  5262.0 2287.71  5278.8 2289.12
#Mann=5,-1,0
  4768.0    0.16       0  4900.6    0.07       0  4931.9    0.16       0
  4993.9    0.07       0  4999.9    0.16       0
Bank Sta=4993.9,4999.9
Exp/Cntr=0.3,0.1

Type RM Length L Ch R = 1,10447,229,229,229
BEGIN DESCRIPTION:
Elm 52 10446.998
END DESCRIPTION:
XS GIS Cut Line= 3
      1513155.02      6767887.99      1513305.61      6767808.05
      1513555.02      6767687.99
#Sta/Elev= 30
  4829.5 2187.58  4903.6 2176.45  4909.3 2178.37  4919.9 2174.64  4925.6 2175.34
  4941.9 2169.50  4947.6 2170.13  4963.9 2166.58  4969.6 2167.64  4982.8 2164.55
  4983.3 2164.05  4988.9 2164.55  5002.4 2165.02  5008.3 2169.69  5013.8 2169.34
  5021.5 2173.38  5030.9 2175.91  5053.5 2180.00  5059.1 2178.73  5110.3 2191.11
  5143.6 2196.91  5188.0 2211.60  5217.4 2229.05  5232.4 2236.32  5240.1 2245.29
  5245.6 2246.82  5262.7 2262.56  5268.2 2265.15  5274.0 2273.37  5276.8 2273.37
#Mann=3,-1,0
  4829.5    0.16       0  4982.8    0.07       0  4988.9    0.16       0
Bank Sta=4982.8,4988.9
Exp/Cntr=0.3,0.1

Type RM Length L Ch R = 1,10218,106,106,106
BEGIN DESCRIPTION:
Elm 52 10217.97
END DESCRIPTION:
XS GIS Cut Line= 3
      1512927.96      6768181.10      1513204.04      6768007.47
      1513594.69      6767797.38
#Sta/Elev= 30
  4671.5 2217.79  4692.1 2211.63  4786.3 2193.05  4816.9 2195.35  4822.8 2193.24
  4853.4 2192.87  4868.7 2189.54  4874.6 2185.01  4881.6 2185.14  4889.9 2186.93
  4895.8 2181.97  4911.1 2184.17  4917.1 2175.61  4926.4 2175.59  4932.3 2168.54
  4947.6 2168.58  4953.6 2164.46  4984.2 2163.60  5001.0 2166.06  5030.0 2162.59
  5030.5 2162.09  5036.7 2162.59  5093.4 2169.71  5109.6 2175.61  5131.5 2179.66
  5219.2 2187.35  5293.9 2197.75  5339.3 2206.85  5383.1 2225.39  5441.2 2260.46
#Mann=4,-1,0
  4671.5    0.07       0  4881.6    0.16       0  5030.0    0.07       0
  5036.7    0.16       0
Bank Sta=5030,5036.7
Exp/Cntr=0.3,0.1

Type RM Length L Ch R = 1,10112,109,109,109
BEGIN DESCRIPTION:
Elm 52 10111.76
END DESCRIPTION:
XS GIS Cut Line= 3
      1513000.94      6768257.45      1513261.33      6768090.80
      1513607.23      6767852.13
#Sta/Elev= 30
  4693.5 2215.27  4703.0 2212.69  4718.2 2216.59  4724.1 2212.94  4733.4 2215.16
  4739.4 2211.59  4756.2 2210.42  4760.5 2209.20  4775.7 2214.37  4812.1 2206.46
  4818.0 2201.71  4833.2 2198.02  4848.4 2200.43  4854.4 2197.81  4863.7 2200.38
  4884.8 2199.57  4890.7 2196.49  4921.2 2194.03  4935.8 2188.93  4971.4 2162.33
  4975.3 2161.74  4975.8 2161.24  4982.0 2161.74  5032.0 2165.65  5065.5 2177.09
  5237.9 2189.47  5316.3 2199.60  5381.9 2216.31  5417.7 2232.15  5422.9 2236.89
#Mann=5,-1,0
  4693.5    0.16       0  4756.2    0.07       0  4975.3    0.07       0
  4982.0    0.07       0  5032.0    0.16       0
Bank Sta=4975.3,4982
Exp/Cntr=0.3,0.1

Type RM Length L Ch R = 1,10003,157,157,157
BEGIN DESCRIPTION:
Elm 52 10003.14
END DESCRIPTION:
XS GIS Cut Line= 3
      1513186.72      6768285.21      1513335.98      6768168.92
      1513646.74      6767868.58
#Sta/Elev= 30
  4809.8 2219.05  4838.9 2219.51  4871.0 2218.86  4884.3 2212.45  4892.4 2204.77
  4898.7 2201.94  4906.9 2195.16  4913.2 2193.23  4927.7 2183.92  4934.4 2177.03
  4942.2 2172.03  4967.9 2165.11  4991.9 2160.47  5016.9 2159.44  5017.4 2158.94
  5023.6 2159.44  5027.2 2161.82  5034.4 2162.64  5048.5 2169.95  5055.5 2176.06
  5133.4 2179.95  5232.4 2188.83  5317.3 2199.99  5345.4 2207.91  5380.9 2224.96
  5387.8 2226.04  5395.0 2231.00  5402.0 2232.34  5428.0 2248.72  5431.2 2248.72
#Mann=5,-1,0
  4809.8    0.16       0  4838.9    0.07       0  4967.9    0.16       0
  5016.9    0.07       0  5023.6    0.16       0
Bank Sta=5016.9,5023.6
Exp/Cntr=0.3,0.1

Type RM Length L Ch R = 1,9846,104,104,104
BEGIN DESCRIPTION:
Elm 52 9846.01
END DESCRIPTION:
XS GIS Cut Line= 3
      1513214.47      6768359.89      1513480.08      6768212.33
      1513679.75      6767917.16
#Sta/Elev= 30
  4696.3 2216.32  4743.3 2215.29  4751.9 2215.49  4787.8 2215.27  4793.5 2212.33
  4815.2 2194.95  4837.0 2179.58  4853.0 2173.26  4858.7 2169.67  4868.5 2168.88
  4880.4 2164.81  4955.9 2160.79  4974.3 2157.00  4974.8 2156.50  4981.0 2157.00
  4993.7 2157.63  4999.4 2166.58  5005.8 2167.47  5014.6 2173.23  5086.5 2176.38
  5128.5 2181.16  5287.3 2208.14  5302.3 2213.63  5308.3 2213.62  5317.2 2217.71
  5323.3 2218.55  5338.2 2227.74  5344.3 2229.38  5353.0 2236.53  5356.5 2236.53
#Mann=5,-1,0
  4696.3    0.16       0  4743.3    0.07       0  4751.9    0.16       0
  4974.3    0.07       0  4981.0    0.16       0
Bank Sta=4974.3,4981
Exp/Cntr=0.3,0.1

Type RM Length L Ch R = 1,9742,97,97,97
BEGIN DESCRIPTION:
Elm 52 9742.44
END DESCRIPTION:
XS GIS Cut Line= 3
      1513242.21      6768399.83      1513520.01      6768306.08
      1513735.29      6767998.78
#Sta/Elev= 30
  4703.2 2209.92  4716.7 2209.37  4728.6 2203.51  4754.7 2200.59  4760.0 2204.93
  4786.2 2199.15  4791.5 2203.02  4817.7 2197.03  4823.0 2200.33  4843.3 2197.19
  4849.1 2194.36  4854.4 2196.11  4875.0 2188.88  4885.9 2179.12  4917.4 2165.92
  4969.7 2160.24  4987.8 2155.83  4988.3 2155.33  4994.5 2155.83  5006.3 2156.42
  5019.2 2162.28  5048.8 2163.23  5063.6 2167.13  5099.4 2172.18  5170.9 2178.28
  5227.5 2188.13  5292.9 2208.01  5343.5 2227.62  5358.3 2231.89  5371.6 2231.58
#Mann=3,-1,0
  4703.2    0.16       0  4987.8    0.07       0  4994.5    0.16       0
Bank Sta=4987.8,4994.5
Exp/Cntr=0.3,0.1

Type RM Length L Ch R = 1,9645,78,78,78
BEGIN DESCRIPTION:
Elm 52 9644.76
END DESCRIPTION:
XS GIS Cut Line= 3
      1513454.06      6768542.16      1513598.13      6768363.37
      1513739.68      6768042.30
#Sta/Elev= 30
  4782.5 2211.05  4793.1 2209.29  4807.5 2213.25  4836.3 2215.63  4857.3 2212.36
  4871.5 2209.87  4877.9 2206.24  4885.9 2204.37  4892.3 2198.43  4935.5 2183.07
  4956.3 2178.32  4978.6 2175.98  4995.5 2165.73  5005.9 2156.62  5011.3 2154.66
  5011.8 2154.16  5018.0 2154.66  5038.0 2159.17  5105.4 2161.70  5136.7 2167.89
  5142.2 2167.35  5149.1 2169.75  5212.1 2178.64  5269.7 2197.16  5287.6 2199.92
  5293.0 2203.26  5310.9 2205.79  5316.4 2209.02  5356.8 2218.47  5363.0 2222.08
#Mann=5,-1,0
  4782.5    0.16       0  4857.3    0.07       0  4995.5    0.16       0
  5011.3    0.07       0  5018.0    0.16       0
Bank Sta=5011.3,5018
Exp/Cntr=0.3,0.1

Type RM Length L Ch R = 1,9567,105,105,105
BEGIN DESCRIPTION:
Elm 52 9567.36
END DESCRIPTION:
XS GIS Cut Line= 3
      1513530.45      6768632.42      1513667.58      6768380.73
      1513782.17      6768033.47
#Sta/Elev= 30
  4721.6 2217.34  4758.8 2213.33  4790.9 2203.23  4808.2 2196.14  4824.3 2191.38
  4865.6 2185.11  4977.2 2172.56  4993.3 2165.24  4999.9 2155.38  5012.8 2154.03
  5013.3 2153.53  5019.6 2154.03  5032.2 2157.07  5084.9 2159.79  5111.4 2163.82
  5116.7 2163.32  5143.2 2171.47  5148.4 2171.69  5174.9 2180.28  5180.2 2179.71
  5200.6 2183.27  5232.2 2190.82  5243.7 2195.46  5263.8 2200.64  5270.2 2205.03
  5301.9 2214.15  5333.7 2221.78  5358.6 2225.99  5365.4 2228.58  5373.9 2228.92
#Mann=5,-1,0
  4721.6    0.16       0  4790.9    0.07       0  4865.6    0.16       0
  5012.8    0.07       0  5019.6    0.16       0
Bank Sta=5012.8,5019.6
Exp/Cntr=0.3,0.1

Type RM Length L Ch R = 1,9462,211,211,211
BEGIN DESCRIPTION:
Elm 52 9461.88
END DESCRIPTION:
XS GIS Cut Line= 3
      1513615.49      6768693.25      1513770.01      6768385.94
      1513842.62      6768081.65
#Sta/Elev= 30
  4658.0 2213.26  4668.5 2212.17  4697.5 2212.97  4713.4 2210.58  4764.6 2188.05
  4790.8 2181.17  4802.7 2179.00  4819.4 2178.69  4959.0 2166.33  5002.0 2157.99
  5017.0 2152.32  5017.5 2151.82  5023.8 2152.32  5045.6 2154.74  5051.3 2157.26
  5092.8 2160.24  5102.7 2162.53  5123.2 2171.44  5129.8 2176.38  5134.9 2175.92
  5164.3 2187.05  5171.9 2188.92  5177.0 2187.45  5214.0 2199.20  5219.1 2198.39
  5236.3 2206.42  5256.1 2212.19  5261.2 2212.22  5267.2 2215.89  5314.8 2225.27
#Mann=5,-1,0
  4658.0    0.16       0  4668.5    0.07       0  4790.8    0.16       0
  5017.0    0.07       0  5023.8    0.16       0
Bank Sta=5017,5023.8
Exp/Cntr=0.3,0.1

Type RM Length L Ch R = 1,9251,138,138,138
BEGIN DESCRIPTION:
Elm 52 9250.66
END DESCRIPTION:
XS GIS Cut Line= 3
      1513648.47      6768688.03      1513940.15      6768488.37
      1514096.41      6768134.18
#Sta/Elev= 30
  4636.5 2210.49  4656.5 2212.53  4668.9 2209.59  4734.6 2179.85  4814.0 2173.13
  4863.2 2167.32  4872.1 2165.34  4878.1 2161.44  4899.1 2158.15  4964.8 2153.65
  4971.6 2151.95  4976.3 2148.94  4976.8 2148.44  4983.2 2148.94  5001.3 2154.44
  5010.6 2159.71  5016.0 2168.15  5114.8 2172.74  5230.8 2181.20  5260.1 2187.59
  5265.6 2187.13  5283.5 2194.15  5288.9 2193.37  5306.8 2201.37  5312.2 2199.97
  5335.6 2212.51  5341.0 2210.05  5358.9 2216.78  5364.3 2213.40  5377.1 2216.14
#Mann=4,-1,0
  4636.5    0.07       0  4814.0    0.16       0  4976.3    0.07       0
  4983.2    0.16       0
Bank Sta=4976.3,4983.2
Exp/Cntr=0.3,0.1

Type RM Length L Ch R = 1,9113,214,214,214
BEGIN DESCRIPTION:
Elm 52 9113.26
END DESCRIPTION:
XS GIS Cut Line= 3
      1513912.38      6768934.53      1514013.07      6768592.53
      1514179.48      6768152.24
#Sta/Elev= 30
  4637.9 2202.58  4655.1 2207.14  4673.7 2207.25  4696.0 2203.02  4707.3 2196.55
  4734.5 2186.36  4759.4 2179.57  4878.3 2169.34  4894.9 2166.08  4916.8 2157.98
  4936.6 2157.71  4985.3 2148.05  4985.8 2147.55  4992.2 2148.05  4994.2 2150.16
  5009.3 2151.45  5020.6 2155.17  5099.8 2153.57  5116.9 2157.85  5124.7 2162.67
  5130.0 2160.65  5154.9 2169.27  5270.2 2175.92  5355.4 2184.82  5373.4 2190.50
  5405.1 2205.56  5416.2 2213.66  5435.3 2221.76  5440.6 2226.70  5465.1 2238.63
#Mann=4,-1,0
  4637.9    0.07       0  4673.7    0.16       0  4985.3    0.07       0
  4992.2    0.16       0
Bank Sta=4985.3,4992.2
Exp/Cntr=0.3,0.1

Type RM Length L Ch R = 1,8899,135,135,135
BEGIN DESCRIPTION:
Elm 52 8899.19
END DESCRIPTION:
XS GIS Cut Line= 3
      1514065.14      6768918.94      1514191.88      6768488.37
      1514238.76      6768193.20
#Sta/Elev= 30
  4550.7 2206.08  4562.1 2204.35  4567.6 2201.00  4572.8 2201.75  4580.1 2199.80
  4600.9 2192.94  4606.2 2194.42  4634.3 2183.03  4639.5 2183.58  4672.8 2173.39
  4687.2 2171.33  4760.2 2165.36  4822.7 2163.51  4906.1 2164.43  4916.5 2163.45
  4921.9 2159.48  4927.1 2159.30  4937.4 2153.41  4993.8 2150.85  5026.8 2144.70
  5027.3 2144.20  5033.7 2144.70  5040.4 2149.78  5048.4 2159.50  5060.7 2165.42
  5172.0 2173.58  5232.8 2204.21  5253.0 2219.98  5293.4 2243.33  5298.4 2243.33
#Mann=4,-1,0
  4550.7    0.07       0  4580.1    0.16       0  5026.8    0.07       0
  5033.7    0.16       0
Bank Sta=5026.8,5033.7
Exp/Cntr=0.3,0.1

Type RM Length L Ch R = 1,8764,206,206,206
BEGIN DESCRIPTION:
Elm 52 8764.05
END DESCRIPTION:
XS GIS Cut Line= 3
      1514127.65      6768859.89      1514311.68      6768535.24
      1514405.05      6768312.17
#Sta/Elev= 30
  4627.3 2195.66  4633.6 2197.31  4649.5 2189.45  4655.3 2190.33  4671.2 2182.90
  4676.9 2182.88  4692.8 2177.60  4698.5 2178.43  4705.4 2176.37  4714.4 2176.21
  4730.3 2170.83  4757.7 2167.18  4876.0 2163.13  4919.3 2155.59  4935.2 2155.66
  5014.4 2143.38  5014.9 2142.88  5021.3 2143.38  5062.5 2154.59  5084.2 2167.04
  5105.9 2177.02  5129.3 2182.73  5147.7 2184.74  5170.9 2190.97  5200.7 2205.05
  5206.1 2206.29  5214.3 2212.86  5224.5 2218.21  5229.9 2219.13  5242.3 2230.46
#Mann=4,-1,0
  4627.3    0.07       0  4705.4    0.16       0  5014.4    0.07       0
  5021.3    0.16       0
Bank Sta=5014.4,5021.3
Exp/Cntr=0.3,0.1

Type RM Length L Ch R = 1,8558,208,208,208
BEGIN DESCRIPTION:
Elm 52 8557.568
END DESCRIPTION:
XS GIS Cut Line= 3
      1514255.02      6768887.97      1514486.92      6768619.05
      1514654.99      6768388.01
#Sta/Elev= 30
  4644.9 2200.29  4652.0 2199.51  4658.6 2195.76  4666.2 2193.96  4672.9 2190.08
  4680.5 2188.27  4687.1 2184.16  4694.8 2182.57  4701.4 2178.97  4723.3 2172.43
  4729.9 2169.02  4801.2 2161.94  4840.0 2159.67  4914.2 2158.49  4942.7 2156.90
  4977.8 2147.43  4993.9 2141.13  4994.4 2140.63  5000.8 2141.13  5050.4 2150.05
  5063.1 2158.54  5077.5 2165.27  5113.0 2173.10  5127.7 2177.96  5149.7 2187.23
  5207.3 2222.59  5222.0 2232.39  5242.8 2248.74  5282.6 2276.02  5285.7 2276.02
#Mann=4,-1,0
  4644.9    0.07       0  4840.0    0.16       0  4993.9    0.07       0
  5000.8    0.16       0
Bank Sta=4993.9,5000.8
Exp/Cntr=0.3,0.1

Type RM Length L Ch R = 1,8350,163,163,163
BEGIN DESCRIPTION:
Elm 52 8349.95
END DESCRIPTION:
XS GIS Cut Line= 3
      1514382.86      6768993.57      1514648.48      6768738.37
      1514799.35      6768552.81
#Sta/Elev= 30
  4627.1 2186.95  4646.6 2177.97  4674.9 2169.90  4689.1 2168.00  4767.0 2163.25
  4844.7 2162.34  4862.8 2158.48  4894.1 2153.10  4972.1 2144.38  4979.0 2145.56
  5011.0 2140.49  5011.5 2139.99  5018.0 2140.49  5028.9 2142.84  5049.7 2157.09
  5072.0 2168.68  5092.8 2176.13  5113.6 2179.61  5121.5 2183.99  5142.3 2190.26
  5156.7 2196.18  5171.1 2206.83  5177.5 2208.45  5185.4 2214.13  5191.9 2215.27
  5199.8 2220.67  5206.3 2221.31  5214.2 2226.12  5220.6 2224.73  5234.6 2233.52
#Mann=4,-1,0
  4627.1    0.07       0  4862.8    0.16       0  5011.0    0.07       0
  5018.0    0.16       0
Bank Sta=5011,5018
Exp/Cntr=0.3,0.1

Type RM Length L Ch R = 1,8187,267,267,267
BEGIN DESCRIPTION:
Elm 52 8186.62
END DESCRIPTION:
XS GIS Cut Line= 3
      1514500.91      6769085.59      1514757.86      6768854.69
      1514889.24      6768642.06
#Sta/Elev= 30
  4658.5 2188.67  4666.6 2184.71  4674.0 2186.49  4680.8 2181.65  4688.2 2182.51
  4695.0 2178.78  4702.4 2178.69  4709.2 2174.88  4716.6 2173.96  4737.6 2166.89
  4857.9 2153.28  4894.0 2147.46  4921.4 2145.44  4949.8 2140.90  4957.3 2137.15
  4964.0 2138.41  4968.0 2135.62  4968.5 2135.12  4975.0 2135.62  4978.3 2138.02
  4985.7 2137.64  5004.0 2141.23  5012.9 2149.13  5028.3 2154.67  5064.9 2157.32
  5101.6 2163.75  5122.8 2165.03  5159.5 2173.05  5217.4 2180.58  5253.9 2189.65
#Mann=4,-1,0
  4658.5    0.07       0  4894.0   0.035       0  4968.0   0.035       0
  4975.0   0.035       0
Bank Sta=4968,4975
Exp/Cntr=0.3,0.1

Type RM Length L Ch R = 1,7920,251,251,251
BEGIN DESCRIPTION:
Elm 52 7919.98
END DESCRIPTION:
XS GIS Cut Line= 3
      1514653.67      6769269.64      1514815.15      6769104.69
      1515020.80      6768724.48
#Sta/Elev= 30
  4764.5 2201.55  4858.5 2197.75  4879.7 2195.01  4886.8 2195.28  4901.0 2187.48
  4908.0 2173.39  4915.1 2165.50  4922.1 2149.39  4936.3 2139.78  4950.4 2136.13
  4961.1 2135.47  4961.6 2134.97  4968.1 2135.47  4991.7 2138.42  5045.2 2140.31
  5088.9 2139.64  5114.9 2141.53  5115.4 2141.61  5154.5 2144.31  5170.7 2150.30
  5176.4 2149.04  5192.6 2154.11  5198.3 2152.46  5207.6 2155.27  5220.2 2156.70
  5258.3 2158.06  5334.6 2166.30  5405.7 2172.73  5421.9 2175.94  5427.6 2175.49
#Mann=6,-1,0
  4764.5    0.07       0  4961.1    0.07       0  4968.1    0.07       0
  5114.9    0.16       0  5115.4    0.07       0  5334.6    0.16       0
Bank Sta=4961.1,4968.1
Exp/Cntr=0.3,0.1

Type RM Length L Ch R = 1,7669,258,258,258
BEGIN DESCRIPTION:
Elm 52 7668.66
END DESCRIPTION:
XS GIS Cut Line= 3
      1514908.89      6769372.06      1515039.11      6769090.80
      1515125.92      6768785.23
#Sta/Elev= 30
  4688.9 2183.98  4695.2 2179.57  4708.5 2176.04  4741.1 2162.38  4748.5 2157.74
  4770.5 2152.18  4781.4 2150.86  4792.6 2147.99  4832.7 2142.45  4838.2 2140.75
  4884.1 2136.44  4924.4 2137.28  4968.9 2136.32  4990.9 2131.93  5001.0 2131.72
  5001.5 2131.22  5008.0 2131.72  5012.1 2134.56  5022.5 2138.39  5032.9 2143.67
  5038.4 2148.65  5043.6 2148.56  5053.7 2151.53  5064.1 2152.91  5152.4 2159.28
  5187.6 2161.82  5223.5 2163.89  5230.5 2165.26  5251.2 2166.17  5316.5 2172.05
#Mann=6,-1,0
  4688.9    0.07       0  4708.5    0.16       0  5001.0    0.07       0
  5008.0    0.16       0  5152.4    0.07       0  5187.6    0.16       0
Bank Sta=5001,5008
Exp/Cntr=0.3,0.1

Type RM Length L Ch R = 1,7411,200,200,200
BEGIN DESCRIPTION:
Elm 52 7410.56
END DESCRIPTION:
XS GIS Cut Line= 3
      1514960.98      6769439.76      1515245.70      6769234.90
      1515273.47      6768972.83
#Sta/Elev= 30
  4644.2 2164.65  4649.8 2164.65  4655.5 2160.20  4661.7 2159.45  4670.3 2155.96
  4676.4 2154.94  4705.9 2147.33  4762.3 2138.61  4791.8 2136.44  4806.5 2134.06
  4821.2 2133.42  4833.9 2134.23  4870.9 2133.25  4883.9 2134.23  4942.8 2133.11
  4957.1 2132.07  4978.4 2132.39  4991.5 2130.80  5008.5 2129.98  5009.0 2129.48
  5015.0 2129.48  5015.5 2129.98  5022.0 2131.42  5031.4 2136.20  5036.4 2141.16
  5042.1 2144.66  5052.2 2149.05  5092.4 2151.63  5134.2 2153.21  5258.5 2161.23
#Mann=3,-1,0
  4644.2    0.16       0  5008.5    0.07       0  5015.5    0.16       0
Bank Sta=5008.5,5015.5
Exp/Cntr=0.3,0.1

Type RM Length L Ch R = 1,7211,196,196,196
BEGIN DESCRIPTION:
Elm 52 7210.94
END DESCRIPTION:
XS GIS Cut Line= 3
      1514903.67      6769543.93      1515256.12      6769385.94
      1515571.96      6769382.49
#Sta/Elev= 30
  4614.6 2192.00  4619.2 2187.87  4636.9 2182.52  4642.4 2178.14  4648.9 2175.79
  4659.9 2174.11  4671.1 2169.34  4681.8 2167.58  4688.8 2165.03  4735.1 2157.54
  4769.5 2149.93  4838.8 2140.49  4862.0 2139.38  4882.7 2136.74  4922.9 2131.89
  4966.7 2132.05  4977.7 2130.52  4979.3 2127.81  4979.8 2127.31  4987.5 2127.81
  5029.7 2128.27  5059.7 2131.44  5069.7 2130.72  5119.7 2140.22  5129.7 2143.19
  5139.7 2144.18  5254.9 2145.62  5299.7 2148.32  5309.7 2150.73  5316.7 2156.15
#Mann=5,-1,0
  4614.6    0.07       0  4882.7    0.16       0  4979.3    0.07       0
  4987.5    0.16       0  5254.9    0.07       0
Bank Sta=4979.3,4987.5
Exp/Cntr=0.3,0.1

Type RM Length L Ch R = 1,7015,261,261,261
BEGIN DESCRIPTION:
Elm 52 7015.32
END DESCRIPTION:
XS GIS Cut Line= 3
      1514976.61      6769722.74      1515270.01      6769576.91
      1515798.31      6769372.52
#Sta/Elev= 30
  4653.0 2195.40  4677.0 2193.90  4716.2 2176.05  4783.4 2158.42  4805.8 2154.65
  4833.8 2154.30  4908.0 2140.14  4946.7 2137.21  5024.8 2125.15  5025.3 2124.65
  5033.0 2125.15  5051.3 2130.10  5125.0 2131.84  5207.4 2141.36  5318.4 2145.22
  5353.8 2156.89  5378.4 2155.32  5383.8 2150.75  5403.0 2153.57  5408.4 2149.91
  5432.9 2156.99  5438.3 2153.34  5457.5 2158.82  5462.9 2156.28  5468.5 2158.79
  5479.2 2157.41  5487.5 2154.30  5492.8 2157.90  5511.4 2153.99  5547.1 2156.72
#Mann=5,-1,0
  4653.0    0.07       0  4946.7    0.16       0  5024.8    0.07       0
  5033.0    0.16       0  5207.4    0.07       0
Bank Sta=5024.8,5033
Exp/Cntr=0.3,0.1

Type RM Length L Ch R = 1,6754,170,170,170
BEGIN DESCRIPTION:
Elm 52 6754.06
END DESCRIPTION:
XS GIS Cut Line= 3
      1515167.62      6769870.30      1515455.77      6769740.10
      1515841.44      6769395.95
#Sta/Elev= 30
  4615.0 2185.81  4623.1 2181.94  4636.1 2172.20  4659.3 2160.61  4676.9 2154.08
  4688.9 2148.29  4705.5 2142.73  4739.8 2139.84  4809.6 2135.77  4826.6 2133.75
  4855.2 2134.04  4872.8 2131.91  4878.3 2129.93  4924.5 2128.99  4946.1 2125.89
  4967.8 2125.04  4984.6 2122.40  4985.1 2121.90  4992.8 2122.40  4996.2 2126.58
  5002.9 2128.45  5010.4 2128.79  5031.3 2133.97  5038.0 2137.05  5072.4 2135.92
  5208.6 2141.63  5278.8 2145.85  5286.3 2145.34  5329.0 2147.29  5448.1 2157.14
#Mann=5,-1,0
  4615.0    0.07       0  4739.8    0.16       0  4984.6    0.07       0
  4992.8    0.16       0  5072.4    0.07       0
Bank Sta=4984.6,4992.8
Exp/Cntr=0.3,0.1

Type RM Length L Ch R = 1,6584,195,195,195
BEGIN DESCRIPTION:
Elm 52 6583.94
END DESCRIPTION:
XS GIS Cut Line= 3
      1515426.23      6770042.22      1515596.40      6769832.12
      1515886.34      6769448.42
#Sta/Elev= 30
  4726.8 2178.28  4729.8 2178.28  4735.7 2175.15  4743.7 2174.44  4750.1 2171.40
  4764.5 2168.36  4778.9 2163.50  4799.7 2158.79  4828.4 2148.79  4842.8 2142.35
  4857.2 2138.71  4899.5 2133.03  4906.8 2130.95  4935.5 2126.67  4970.7 2126.02
  4985.1 2123.18  4987.4 2120.69  4987.9 2120.19  4995.6 2120.69  5000.2 2121.00
  5014.2 2126.04  5025.7 2127.02  5035.0 2127.71  5049.6 2126.85  5064.1 2128.37
  5070.4 2130.25  5153.7 2138.60  5214.0 2138.92  5305.6 2141.96  5478.1 2155.61
#Mann=5,-1,0
  4726.8    0.07       0  4987.4    0.07       0  4995.6    0.07       0
  5025.7    0.16       0  5153.7    0.07       0
Bank Sta=4987.4,4995.6
Exp/Cntr=0.3,0.1

Type RM Length L Ch R = 1,6389,227,227,227
BEGIN DESCRIPTION:
Elm 52 6388.91
END DESCRIPTION:
XS GIS Cut Line= 3
      1515558.23      6770135.91      1515747.44      6769943.23
      1515993.16      6769491.60
#Sta/Elev= 30
  4724.1 2166.91  4741.5 2161.80  4777.0 2155.60  4805.3 2145.12  4819.3 2143.65
  4833.4 2145.37  4847.6 2144.67  4861.7 2140.88  4890.0 2129.24  4897.1 2127.94
  4911.3 2129.05  4946.6 2125.23  4953.7 2121.82  4960.7 2122.52  4963.7 2119.61
  4964.2 2119.11  4972.0 2119.61  4982.0 2121.40  4994.2 2121.00  4997.0 2123.02
  5003.3 2121.88  5024.5 2124.67  5068.4 2125.01  5128.0 2132.25  5147.2 2138.06
  5159.5 2138.50  5171.7 2135.20  5187.9 2134.76  5231.6 2136.72  5508.3 2157.75
#Mann=5,-1,0
  4724.1    0.07       0  4963.7    0.07       0  4972.0    0.07       0
  5003.3    0.16       0  5147.2    0.07       0
Bank Sta=4963.7,4972
Exp/Cntr=0.3,0.1

Type RM Length L Ch R = 1,6162,232,232,232
BEGIN DESCRIPTION:
Elm 52 6162.18
END DESCRIPTION:
XS GIS Cut Line= 3
      1515613.74      6770198.45      1515896.75      6770047.40
      1516434.94      6769783.51
#Sta/Elev= 30
  4670.7 2167.49  4694.8 2161.93  4723.9 2151.33  4740.1 2148.56  4745.9 2146.12
  4767.9 2142.72  4784.1 2137.34  4796.8 2134.67  4887.5 2134.08  4915.9 2129.04
  4921.5 2126.50  4948.3 2123.35  4981.7 2122.09  4991.5 2120.36  4994.1 2114.83
  4994.6 2114.33  5002.6 2114.83  5003.9 2116.17  5020.8 2117.38  5026.4 2116.62
  5043.3 2120.27  5071.4 2123.42  5116.3 2125.84  5138.8 2125.73  5212.3 2133.82
  5324.0 2143.78  5453.8 2156.84  5477.3 2157.40  5543.7 2166.26  5590.9 2170.78
#Mann=6,-1,0
  4670.7    0.07       0  4948.3    0.16       0  4994.1    0.07       0
  5002.6    0.16       0  5324.0   0.035       0  5477.3    0.07       0
Bank Sta=4994.1,5002.6
Exp/Cntr=0.3,0.1
