--- Elm 63.prj (project) ---

Proj Title=Elm 63 Base Level Engineering
Current Plan=p01
Default Exp/Contr=0.3,0.1
English Units
Geom File=g01
Flow File=f01
Plan File=p01
BEGIN DESCRIPTION:
Elm 63
END DESCRIPTION:

--- Elm 63.p01 (plan) ---

Plan Title=Multiple Run
Short Identifier=Multiple
Geom File=g01
Flow File=f01
Subcritical Flow
K Sum by GR= 0
Std Step Tol= 0.01
Critical Tol= 0.01
Num of Std Step Trials= 20
Max Error Tol= 0.3
Flow Tol Ratio= 0.001
Split Flow NTrial= 30
Split Flow Tol= 0.02
Split Flow Ratio= 0.02
Log Output Level= 0
Friction Slope Method= 1
Unsteady Friction Slope Method= 2
Unsteady Bridges Friction Slope Method= 1
Parabolic Critical Depth
Global Vel Dist=  1 , 1 , 1
Global Log Level= 0
CheckData=True
Encroach Param= -1, 0, 0, 0
BEGIN DESCRIPTION:
Multiple Run
END DESCRIPTION:

--- Elm 63.f01 (steady flow) ---

Flow Title=Multiple
Number of Profiles=7
Profile Names=10-year,25-year,50-year,1pct_min,100-year,1pct_plu,500-year
River Rch & RM= Elm 63,Reach-1,2030
      54      69      80      58      93     129     128
Boundary for River Rch & Prof#=Elm 63,Reach-1,1
Up Type=0
Dn Type=3
Dn Slope=0.005
Boundary for River Rch & Prof#=Elm 63,Reach-1,2
Up Type=0
Dn Type=3
Dn Slope=0.005
Boundary for River Rch & Prof#=Elm 63,Reach-1,3
Up Type=0
Dn Type=3
Dn Slope=0.005
Boundary for River Rch & Prof#=Elm 63,Reach-1,4
Up Type=0
Dn Type=3
Dn Slope=0.005
Boundary for River Rch & Prof#=Elm 63,Reach-1,5
Up Type=0
Dn Type=3
Dn Slope=0.005
Boundary for River Rch & Prof#=Elm 63,Reach-1,6
Up Type=0
Dn Type=3
Dn Slope=0.005
Boundary for River Rch & Prof#=Elm 63,Reach-1,7
Up Type=0
Dn Type=3
Dn Slope=0.005

--- Elm 63.g01 (geometry) ---

Geom Title=Existing Conditions

River Reach=Elm 63,Reach-1
Reach XY= 30
      1520755.00      6769488.00      1521028.13      6769761.83
      1521052.55      6769782.54      1521084.82      6769788.43
      1521370.18      6769787.57      1521399.06      6769790.26
      1521414.65      6769798.85      1521456.60      6769834.14
      1521553.42      6769841.83      1521602.82      6769881.88
      1521657.20      6769894.08      1521702.80      6769931.92
      1521757.20      6769944.08      1521806.74      6769983.81
      1521857.29      6769993.85      1521941.69      6770074.60
      1521965.44      6770086.95      1522170.20      6770088.49
      1522199.14      6770085.94      1522221.75      6770071.54
      1522298.98      6769996.19      1522311.09      6769990.56
      1522353.60      6769984.13      1522372.15      6769971.54
      1522394.70      6769948.11      1522403.12      6769932.29
      1522405.16      6769858.09      1522397.17      6769831.87
      1522358.65      6769786.49      1522355.00      6769738.00

Type RM Length L Ch R = 1,2030,29,29,29
BEGIN DESCRIPTION:
Elm 63 4972
END DESCRIPTION:
XS GIS Cut Line= 3
      1520743.61      6769652.46      1520831.44      6769564.63
      1520909.63      6769483.19
#Sta/Elev= 30
  4875.8 2194.73  4894.1 2195.78  4901.1 2197.66  4908.2 2197.21  4915.3 2197.83
  4936.5 2184.28  4943.6 2180.13  4950.6 2177.75  4957.7 2176.43  4971.5 2175.30
  4978.9 2175.90  4984.0 2174.13  4984.2 2173.63  4987.7 2173.63  4988.0 2174.13
  4993.1 2175.28  5021.5 2176.10  5028.4 2176.79  5035.6 2179.60  5042.5 2180.98
  5049.8 2184.51  5056.7 2184.26  5063.9 2187.45  5070.9 2186.77  5078.1 2189.93
  5085.0 2187.68  5092.2 2190.96  5099.2 2190.71  5106.1 2193.15  5112.9 2193.15
#Mann=4,-1,0
  4875.8    0.07       0  4971.5    0.16       0  4984.0    0.07       0
  4988.0    0.16       0
Bank Sta=4984,4988
Exp/Cntr=0.3,0.1

Type RM Length L Ch R = 1,2001,45,45,45
BEGIN DESCRIPTION:
Elm 63 4996
END DESCRIPTION:
XS GIS Cut Line= 3
      1520778.93      6769646.98      1520851.54      6769584.79
      1520920.62      6769514.85
#Sta/Elev= 30
  4904.4 2197.28  4908.2 2195.30  4914.7 2195.00  4922.4 2190.30  4936.7 2183.58
  4943.3 2179.69  4951.0 2177.12  4957.6 2176.42  4963.5 2175.32  4971.8 2173.68
  4976.4 2173.35  4976.7 2172.85  4980.2 2172.85  4980.4 2173.35  4986.1 2173.40
  4992.7 2174.08  4999.0 2174.15  5007.3 2175.01  5014.3 2174.49  5021.4 2174.94
  5028.4 2174.36  5035.6 2175.86  5042.6 2175.84  5049.7 2177.12  5056.7 2177.98
  5063.9 2180.08  5073.6 2183.57  5085.0 2186.98  5092.1 2188.01  5098.3 2190.74
#Mann=5,-1,0
  4904.4    0.07       0  4963.5    0.16       0  4976.4    0.07       0
  4980.4    0.16       0  5073.6    0.07       0
Bank Sta=4976.4,4980.4
Exp/Cntr=0.3,0.1

Type RM Length L Ch R = 1,1956,37,37,37
BEGIN DESCRIPTION:
Elm 63 4995
END DESCRIPTION:
XS GIS Cut Line= 3
      1520779.78      6769670.44      1520883.61      6769616.95
      1520953.36      6769539.40
#Sta/Elev= 30
  4883.2 2194.82  4897.1 2190.38  4902.7 2191.48  4911.6 2188.75  4919.2 2185.88
  4924.9 2185.38  4934.1 2182.70  4941.4 2179.41  4951.1 2176.41  4963.6 2172.76
  4977.1 2171.54  4977.3 2171.04  4980.8 2171.04  4981.1 2171.54  4985.7 2171.79
  4991.4 2173.04  5014.2 2172.59  5021.6 2172.89  5028.4 2172.42  5042.6 2172.71
  5050.0 2174.64  5056.8 2175.80  5064.2 2179.50  5071.0 2181.64  5080.8 2185.38
  5085.2 2186.51  5092.6 2189.75  5099.4 2190.71  5101.9 2193.53  5104.3 2193.53
#Mann=5,-1,0
  4883.2    0.07       0  4951.1    0.16       0  4977.1    0.07       0
  4981.1    0.16       0  5080.8    0.07       0
Bank Sta=4977.1,4981.1
Exp/Cntr=0.3,0.1

Type RM Length L Ch R = 1,1919,14,14,14
BEGIN DESCRIPTION:
Elm 63 4971
END DESCRIPTION:
XS GIS Cut Line= 3
      1520783.79      6769696.92      1520909.46      6769642.86
      1520967.19      6769563.42
#Sta/Elev= 30
  4863.2 2190.70  4866.6 2190.70  4871.5 2186.76  4877.0 2188.19  4886.3 2185.49
  4895.1 2181.64  4900.5 2183.49  4918.6 2178.03  4924.1 2179.99  4929.8 2176.08
  4940.2 2173.49  4947.6 2172.14  4953.0 2172.61  4962.5 2171.17  4976.6 2171.32
  4992.7 2170.31  4992.9 2169.81  4996.4 2169.81  4996.7 2170.31  5006.6 2170.42
  5015.1 2171.23  5021.2 2170.72  5029.7 2171.22  5035.9 2170.86  5056.8 2172.36
  5071.5 2175.21  5080.0 2179.52  5086.2 2180.41  5092.3 2184.31  5098.2 2184.31
#Mann=4,-1,0
  4863.2    0.07       0  4940.2    0.16       0  4992.7    0.07       0
  4996.7    0.16       0
Bank Sta=4992.7,4996.7
Exp/Cntr=0.3,0.1

Type RM Length L Ch R = 1,1905,30,30,30
BEGIN DESCRIPTION:
Elm 63 4994
END DESCRIPTION:
XS GIS Cut Line= 3
      1520820.58      6769708.63      1520919.16      6769652.58
      1520988.45      6769581.60
#Sta/Elev= 30
  4886.6 2181.84  4892.0 2181.84  4897.7 2180.85  4903.5 2177.71  4913.6 2176.25
  4926.2 2173.97  4936.3 2173.38  4956.8 2170.60  4962.6 2170.86  4978.4 2169.90
  4984.2 2170.11  4992.3 2169.84  4992.6 2169.34  4996.1 2169.34  4996.3 2169.84
  4999.6 2170.03  5007.3 2169.86  5014.5 2170.37  5021.4 2170.04  5028.6 2170.59
  5035.6 2169.94  5042.7 2170.51  5049.7 2169.99  5056.9 2171.29  5063.9 2171.12
  5071.0 2173.37  5078.0 2174.91  5085.2 2177.62  5092.2 2179.55  5099.2 2184.28
#Mann=4,-1,0
  4886.6    0.07       0  4936.3    0.16       0  4992.3    0.07       0
  4996.3    0.16       0
Bank Sta=4992.3,4996.3
Exp/Cntr=0.3,0.1

Type RM Length L Ch R = 1,1875,27,27,27
BEGIN DESCRIPTION:
Elm 63 4993
END DESCRIPTION:
XS GIS Cut Line= 3
      1520850.96      6769723.39      1520940.83      6769674.31
      1521002.00      6769621.83
#Sta/Elev= 28
  4897.6 2185.86  4903.2 2182.16  4913.6 2179.53  4919.3 2176.09  4925.0 2174.98
  4927.4 2174.62  4935.4 2173.40  4941.1 2171.58  4947.8 2170.26  4957.2 2169.55
  4962.9 2169.89  4979.1 2169.03  4984.8 2169.27  4999.5 2168.25  5007.0 2168.72
  5012.7 2168.17  5013.0 2167.67  5016.5 2167.67  5016.7 2168.17  5021.3 2168.43
  5029.0 2168.17  5035.6 2168.44  5043.3 2168.19  5049.8 2168.78  5057.5 2168.69
  5065.0 2169.49  5078.4 2171.28  5080.6 2171.16
#Mann=5,-1,0
  4897.6    0.07       0  4927.4    0.16       0  5012.7    0.07       0
  5016.7    0.16       0  5065.0    0.07       0
Bank Sta=5012.7,5016.7
Exp/Cntr=0.3,0.1

Type RM Length L Ch R = 1,1848,21,21,21
BEGIN DESCRIPTION:
Elm 63 1847.707
END DESCRIPTION:
XS GIS Cut Line= 3
      1520855.04      6769737.98      1520959.84      6769693.38
      1521027.90      6769637.27
#Sta/Elev= 30
  4886.1 2187.50  4888.8 2187.50  4895.2 2183.88  4900.6 2181.92  4907.8 2178.67
  4919.2 2175.10  4924.2 2172.30  4929.7 2171.59  4940.4 2168.96  4947.9 2168.73
  4953.3 2168.94  4962.1 2168.78  4971.5 2167.91  4976.9 2168.25  4994.7 2167.00
  5000.0 2166.85  5006.9 2167.38  5014.7 2166.56  5037.9 2166.67  5043.4 2166.52
  5049.9 2166.62  5055.8 2166.30  5056.0 2165.80  5059.5 2165.80  5059.8 2166.30
  5064.2 2167.70  5071.5 2168.27  5078.6 2170.01  5083.7 2172.44  5088.2 2172.44
#Mann=5,-1,0
  4886.1    0.07       0  4919.2    0.16       0  5037.9    0.07       0
  5055.8    0.07       0  5059.8    0.07       0
Bank Sta=5055.8,5059.8
Exp/Cntr=0.3,0.1

Type RM Length L Ch R = 1,1827,17,17,17
BEGIN DESCRIPTION:
Elm 63 1827.37
END DESCRIPTION:
XS GIS Cut Line= 3
      1520906.54      6769754.62      1520974.22      6769707.77
      1521040.39      6769653.33
#Sta/Elev= 26
  4917.7 2173.81  4921.2 2172.11  4936.1 2167.58  4942.2 2167.53  4951.0 2166.95
  4957.0 2167.62  4971.9 2165.62  4978.0 2166.19  4986.8 2166.21  4992.9 2166.47
  5003.8 2166.46  5005.5 2163.82  5005.8 2163.32  5009.3 2163.32  5009.5 2163.82
  5014.0 2165.72  5018.3 2165.30  5021.9 2164.95  5028.3 2165.79  5036.2 2165.30
  5042.7 2165.77  5050.5 2165.14  5057.0 2165.54  5064.9 2165.38  5078.7 2168.08
  5085.7 2171.26
#Mann=4,-1,0
  4917.7    0.16       0  5005.5    0.07       0  5009.5    0.16       0
  5018.3    0.07       0
Bank Sta=5005.5,5009.5
Exp/Cntr=0.3,0.1

Type RM Length L Ch R = 1,1810,16,16,16
BEGIN DESCRIPTION:
Elm 63 1810.13
END DESCRIPTION:
XS GIS Cut Line= 3
      1520917.82      6769767.65      1520988.98      6769718.19
      1521048.01      6769656.55
#Sta/Elev= 30
  4916.5 2173.43  4921.9 2171.37  4928.0 2169.75  4936.7 2168.04  4942.8 2167.22
  4957.7 2166.80  4963.8 2166.14  4972.5 2160.94  4978.6 2164.36  4986.1 2160.58
  4993.5 2159.73  4998.9 2163.43  5001.6 2163.43  5003.2 2163.43  5007.5 2158.38
  5012.7 2157.61  5013.0 2157.11  5016.5 2157.11  5016.7 2157.61  5021.6 2164.25
  5028.9 2164.89  5035.8 2164.38  5043.0 2164.81  5049.9 2164.80  5057.2 2165.12
  5064.1 2164.95  5071.3 2165.63  5078.2 2166.75  5084.0 2169.63  5088.5 2169.63
#Mann=4,-1,0
  4916.5    0.16       0  5001.6    0.07       0  5012.7    0.07       0
  5016.7    0.07       0
Bank Sta=5012.7,5016.7
Exp/Cntr=0.3,0.1

Type RM Length L Ch R = 1,1794,22,22,22
BEGIN DESCRIPTION:
Elm 63 1794.35
END DESCRIPTION:
XS GIS Cut Line= 3
      1520922.17      6769792.82      1520995.92      6769732.94
      1521049.95      6769673.00
#Sta/Elev= 30
  4902.6 2172.89  4907.6 2172.89  4915.4 2170.42  4921.9 2170.31  4929.8 2168.62
  4936.2 2168.32  4950.6 2166.09  4957.8 2165.49  4965.0 2165.14  4971.4 2160.67
  4979.4 2156.04  4985.8 2155.96  4986.2 2155.82  4991.7 2153.85  4992.0 2153.35
  4995.5 2153.35  4995.7 2153.85  4997.6 2157.59  5000.6 2157.59  5007.3 2154.29
  5014.8 2156.11  5021.5 2159.15  5029.0 2163.83  5035.7 2163.58  5043.2 2164.14
  5049.9 2164.10  5057.4 2164.59  5064.1 2163.81  5071.6 2164.58  5078.3 2167.70
#Mann=4,-1,0
  4902.6    0.16       0  4986.2    0.07       0  4991.7    0.07       0
  4995.7    0.07       0
Bank Sta=4991.7,4995.7
Exp/Cntr=0.3,0.1

Type RM Length L Ch R = 1,1772,32,32,32
BEGIN DESCRIPTION:
Elm 63 1771.66
END DESCRIPTION:
XS GIS Cut Line= 3
      1520945.58      6769818.00      1521011.55      6769750.30
      1521056.00      6769681.91
#Sta/Elev= 30
  4901.8 2168.66  4905.0 2168.66  4908.5 2167.21  4915.6 2167.28  4922.6 2165.82
  4929.7 2165.91  4936.8 2166.38  4943.7 2165.12  4950.9 2165.35  4957.9 2164.67
  4965.0 2165.36  4972.0 2164.10  4979.2 2157.99  4986.2 2156.61  4990.2 2152.41
  4993.3 2149.15  4994.3 2148.57  4994.6 2148.07  4998.1 2148.07  4998.3 2148.57
  5000.7 2148.57  5008.4 2151.04  5014.4 2159.68  5022.9 2159.87  5029.5 2163.37
  5044.7 2163.57  5050.6 2163.30  5058.7 2163.72  5071.7 2163.97  5077.9 2165.84
#Mann=4,-1,0
  4901.8    0.16       0  4990.2    0.07       0  4994.3    0.07       0
  4998.3    0.07       0
Bank Sta=4994.3,4998.3
Exp/Cntr=0.3,0.1

Type RM Length L Ch R = 1,1740,24,24,24
BEGIN DESCRIPTION:
Elm 63 1740.13
END DESCRIPTION:
XS GIS Cut Line= 3
      1520968.13      6769849.28      1521036.72      6769768.53
      1521072.30      6769675.67
#Sta/Elev= 30
  4894.5 2167.27  4900.1 2166.68  4907.8 2166.53  4928.6 2165.21  4935.5 2164.29
  4942.9 2164.32  4949.5 2160.54  4957.2 2158.40  4963.8 2155.15  4971.5 2154.95
  4978.0 2148.71  4985.8 2150.46  4992.3 2145.83  4995.5 2144.72  4995.8 2144.22
  4999.3 2144.22  4999.5 2144.72  5003.4 2144.72  5008.0 2149.21  5013.3 2149.92
  5014.2 2150.72  5022.4 2157.98  5032.7 2162.49  5038.0 2160.58  5043.9 2161.89
  5062.7 2162.66  5068.1 2162.24  5086.7 2164.92  5092.8 2166.60  5099.9 2166.90
#Mann=4,-1,0
  4894.5    0.16       0  4995.5    0.07       0  4999.5    0.16       0
  5014.2    0.07       0
Bank Sta=4995.5,4999.5
Exp/Cntr=0.3,0.1

Type RM Length L Ch R = 1,1716,24,24,24
BEGIN DESCRIPTION:
Elm 63 1715.71
END DESCRIPTION:
XS GIS Cut Line= 3
      1521021.95      6769854.50      1521055.82      6769783.29
      1521085.34      6769688.64
#Sta/Elev= 30
  4921.5 2166.90  4937.2 2165.28  4942.8 2165.81  4950.8 2164.78  4960.0 2161.92
  4965.5 2163.24  4973.0 2159.40  4975.2 2157.33  4982.7 2150.28  4988.2 2151.85
  4995.0 2140.50  5000.4 2140.50  5005.9 2138.97  5012.8 2141.01  5016.0 2137.27
  5016.3 2136.77  5019.8 2136.77  5020.0 2137.27  5026.8 2146.07  5028.7 2147.33
  5037.3 2153.04  5045.3 2157.55  5050.5 2154.57  5058.3 2156.26  5068.7 2161.29
  5077.8 2162.09  5083.0 2161.48  5089.7 2162.84  5097.2 2164.66  5099.5 2164.66
#Mann=5,-1,0
  4921.5    0.07       0  4975.2    0.16       0  5016.0    0.07       0
  5020.0    0.16       0  5028.7    0.07       0
Bank Sta=5016,5020
Exp/Cntr=0.3,0.1

Type RM Length L Ch R = 1,1692,28,28,28
BEGIN DESCRIPTION:
Elm 63 1691.62
END DESCRIPTION:
XS GIS Cut Line= 3
      1521061.02      6769856.23      1521079.25      6769787.63
      1521103.56      6769694.74
#Sta/Elev= 28
  4929.4 2176.54  4937.9 2174.71  4948.3 2171.40  4958.6 2166.90  4964.1 2162.70
  4969.2 2162.37  4979.3 2158.14  4989.7 2153.28  4997.6 2145.27  5000.4 2145.27
  5004.2 2145.56  5010.3 2140.66  5018.7 2135.66  5018.9 2135.16  5022.4 2135.16
  5022.7 2135.66  5031.0 2137.10  5031.5 2137.56  5035.4 2141.16  5039.5 2144.95
  5044.7 2139.35  5051.7 2149.65  5062.0 2159.09  5072.4 2160.40  5079.9 2161.88
  5085.1 2160.74  5092.1 2162.02  5096.4 2162.02
#Mann=5,-1,0
  4929.4    0.07       0  5018.7    0.07       0  5022.7    0.07       0
  5031.5    0.16       0  5035.4    0.07       0
Bank Sta=5018.7,5022.7
Exp/Cntr=0.3,0.1

Type RM Length L Ch R = 1,1664,31,31,31
BEGIN DESCRIPTION:
Elm 63 1663.6
END DESCRIPTION:
XS GIS Cut Line= 3
      1521099.22      6769849.25      1521107.03      6769789.37
      1521118.23      6769702.37
#Sta/Elev= 25
  4938.6 2175.55  4941.6 2175.55  4944.8 2173.27  4949.9 2169.11  4960.0 2164.54
  4970.1 2161.09  4980.2 2158.26  4990.3 2145.87  4997.2 2142.93  5002.2 2142.93
  5010.5 2141.91  5018.9 2135.67  5021.4 2133.30  5021.9 2132.83  5022.2 2132.33
  5025.7 2132.33  5025.9 2132.83  5030.6 2137.18  5040.7 2143.51  5050.8 2155.46
  5060.9 2158.76  5068.9 2159.10  5070.9 2159.18  5081.0 2160.53  5086.7 2162.31
#Mann=5,-1,0
  4938.6    0.07       0  5021.4    0.16       0  5021.9    0.07       0
  5025.9    0.16       0  5068.9    0.07       0
Bank Sta=5021.9,5025.9
Exp/Cntr=0.3,0.1

Type RM Length L Ch R = 1,1633,18,18,18
BEGIN DESCRIPTION:
Elm 63 1632.66
END DESCRIPTION:
XS GIS Cut Line= 3
      1521131.33      6769842.35      1521138.28      6769786.76
      1521147.83      6769696.49
#Sta/Elev= 23
  4945.5 2162.66  4950.2 2162.66  4960.0 2160.79  4970.0 2158.99  4980.1 2157.77
  4990.2 2147.99  4998.4 2140.12  5001.5 2140.12  5009.0 2133.71  5010.3 2132.60
  5016.6 2133.90  5019.6 2131.84  5019.9 2131.34  5023.4 2131.34  5023.6 2131.84
  5030.4 2138.67  5040.5 2144.66  5050.6 2156.19  5060.6 2157.59  5070.7 2158.05
  5080.7 2158.85  5089.0 2161.49  5092.3 2161.49
#Mann=4,-1,0
  4945.5    0.07       0  5009.0    0.16       0  5019.6    0.07       0
  5023.6    0.16       0
Bank Sta=5019.6,5023.6
Exp/Cntr=0.3,0.1

Type RM Length L Ch R = 1,1615,16,16,16
BEGIN DESCRIPTION:
Elm 63 1614.76
END DESCRIPTION:
XS GIS Cut Line= 3
      1521152.17      6769843.18      1521155.64      6769791.97
      1521164.18      6769701.50
#Sta/Elev= 22
  4944.9 2164.94  4950.1 2161.27  4960.1 2158.94  4970.1 2157.89  4980.2 2156.80
  4990.2 2151.82  4995.7 2143.05  5000.7 2143.05  5001.7 2141.96  5010.3 2132.62
  5018.3 2131.78  5018.6 2131.28  5022.1 2131.28  5022.3 2131.78  5030.4 2134.48
  5039.0 2141.55  5044.0 2144.44  5050.4 2156.47  5060.5 2156.62  5070.5 2156.87
  5080.6 2158.46  5087.1 2160.32
#Mann=4,-1,0
  4944.9    0.07       0  5001.7    0.16       0  5018.3    0.07       0
  5022.3    0.16       0
Bank Sta=5018.3,5022.3
Exp/Cntr=0.3,0.1

Type RM Length L Ch R = 1,1599,31,31,31
BEGIN DESCRIPTION:
Elm 63 1598.66
END DESCRIPTION:
XS GIS Cut Line= 3
      1521168.66      6769841.46      1521172.14      6769787.63
      1521176.40      6769711.69
#Sta/Elev= 22
  4946.6 2161.37  4950.8 2161.37  4960.1 2158.22  4966.2 2157.23  4971.2 2156.05
  4980.1 2154.75  4990.1 2149.68  4995.0 2144.90  4997.8 2142.17  5000.5 2142.17
  5002.9 2142.17  5010.2 2134.90  5018.2 2128.49  5018.5 2127.99  5022.0 2127.99
  5022.2 2128.49  5030.2 2134.09  5040.2 2144.62  5050.2 2151.01  5060.3 2156.43
  5070.3 2157.13  5076.6 2159.02
#Mann=4,-1,0
  4946.6    0.07       0  4995.0    0.16       0  5018.2    0.07       0
  5022.2    0.16       0
Bank Sta=5018.2,5022.2
Exp/Cntr=0.3,0.1

Type RM Length L Ch R = 1,1568,32,32,32
BEGIN DESCRIPTION:
Elm 63 1568.07
END DESCRIPTION:
XS GIS Cut Line= 3
      1521199.92      6769850.11      1521202.52      6769791.97
      1521205.97      6769712.55
#Sta/Elev= 21
  4937.9 2157.05  4942.4 2155.53  4950.0 2154.62  4960.0 2154.00  4970.0 2152.65
  4980.1 2146.76  4982.2 2145.55  4990.1 2141.01  4995.6 2134.08  5000.6 2134.08
  5008.1 2127.88  5008.3 2127.38  5011.8 2127.38  5012.1 2127.88  5020.1 2130.59
  5030.1 2137.93  5040.1 2143.64  5050.1 2150.51  5060.1 2154.50  5070.1 2155.95
  5075.6 2157.82
#Mann=4,-1,0
  4937.9    0.07       0  4982.2    0.16       0  5008.1    0.07       0
  5012.1    0.16       0
Bank Sta=5008.1,5012.1
Exp/Cntr=0.3,0.1

Type RM Length L Ch R = 1,1536,23,23,23
BEGIN DESCRIPTION:
Elm 63 1536.18
END DESCRIPTION:
XS GIS Cut Line= 3
      1521232.90      6769849.26      1521234.64      6769785.89
      1521243.97      6769711.26
#Sta/Elev= 22
  4938.7 2154.41  4941.8 2154.41  4950.0 2153.10  4960.0 2152.51  4968.7 2151.85
  4970.0 2151.75  4980.0 2147.63  4990.0 2141.88  4998.5 2132.92  5002.1 2132.92
  5008.0 2124.32  5008.3 2123.82  5011.8 2123.82  5012.0 2124.32  5020.1 2131.29
  5030.2 2142.98  5040.3 2152.19  5045.3 2153.36  5050.4 2153.81  5060.4 2158.35
  5070.5 2161.41  5077.3 2163.85
#Mann=4,-1,0
  4938.7    0.07       0  4968.7    0.16       0  5008.0    0.07       0
  5012.0    0.16       0
Bank Sta=5008,5012
Exp/Cntr=0.3,0.1

Type RM Length L Ch R = 1,1513,24,24,24
BEGIN DESCRIPTION:
Elm 63 1513.12
END DESCRIPTION:
XS GIS Cut Line= 3
      1521246.79      6769858.79      1521258.07      6769785.03
      1521259.80      6769712.56
#Sta/Elev= 24
  4928.3 2154.36  4931.2 2154.36  4939.2 2153.41  4946.9 2152.21  4951.9 2151.56
  4959.4 2150.98  4960.7 2150.57  4969.6 2147.74  4979.7 2143.93  4989.8 2138.94
  4998.9 2128.47  5002.9 2128.47  5007.9 2124.79  5008.2 2124.29  5011.7 2124.29
  5011.9 2124.79  5019.9 2130.13  5030.0 2137.79  5040.0 2147.06  5050.0 2154.54
  5050.1 2154.59  5060.0 2159.06  5070.0 2162.91  5075.4 2166.04
#Mann=5,-1,0
  4928.3    0.07       0  4960.7    0.16       0  5007.9    0.07       0
  5011.9    0.16       0  5050.1    0.07       0
Bank Sta=5007.9,5011.9
Exp/Cntr=0.3,0.1

Type RM Length L Ch R = 1,1489,24,24,24
BEGIN DESCRIPTION:
Elm 63 1489
END DESCRIPTION:
XS GIS Cut Line= 3
      1521266.76      6769860.51      1521281.51      6769789.37
      1521292.79      6769718.21
#Sta/Elev= 26
  4925.8 2152.05  4929.6 2152.05  4937.6 2151.02  4942.7 2149.74  4948.8 2149.12
  4951.5 2149.16  4959.0 2149.28  4969.2 2147.88  4979.4 2139.18  4987.8 2132.93
  4992.9 2127.81  4994.6 2123.51  4994.8 2123.01  4998.3 2123.01  4998.6 2123.51
  5001.7 2123.51  5006.5 2125.32  5010.0 2126.64  5020.1 2133.73  5030.2 2143.15
  5040.3 2149.79  5049.0 2151.89  5054.1 2151.08  5060.6 2153.30  5068.1 2157.15
  5070.5 2157.15
#Mann=5,-1,0
  4925.8    0.07       0  4951.5    0.16       0  4994.6    0.07       0
  4998.6    0.16       0  5006.5    0.07       0
Bank Sta=4994.6,4998.6
Exp/Cntr=0.3,0.1

Type RM Length L Ch R = 1,1465,21,21,21
BEGIN DESCRIPTION:
Elm 63 1464.79
END DESCRIPTION:
XS GIS Cut Line= 3
      1521271.11      6769874.40      1521305.82      6769788.50
      1521323.18      6769703.40
#Sta/Elev= 30
  4906.6 2151.98  4913.5 2151.22  4924.3 2151.03  4930.0 2149.74  4935.4 2149.25
  4942.9 2148.69  4945.9 2148.46  4954.1 2148.86  4959.5 2148.25  4967.4 2147.91
  4977.3 2134.23  4978.2 2132.99  4983.7 2125.89  4989.1 2126.10  4994.8 2122.60
  4995.1 2122.10  4998.6 2122.10  4998.8 2122.60  5002.1 2122.60  5010.0 2127.11
  5017.6 2132.42  5022.7 2132.61  5030.4 2142.88  5040.6 2147.78  5050.8 2149.69
  5061.0 2151.48  5068.1 2154.50  5073.2 2154.38  5081.2 2158.80  5086.1 2158.80
#Mann=5,-1,0
  4906.6    0.07       0  4942.9    0.16       0  4977.3    0.07       0
  4994.8    0.07       0  4998.8    0.07       0
Bank Sta=4994.8,4998.8
Exp/Cntr=0.3,0.1

Type RM Length L Ch R = 1,1444,19,19,19
BEGIN DESCRIPTION:
Elm 63 1444.21
END DESCRIPTION:
XS GIS Cut Line= 3
      1521291.93      6769854.46      1521328.39      6769784.16
      1521344.87      6769715.60
#Sta/Elev= 27
  4924.8 2148.53  4932.1 2147.85  4934.7 2147.85  4940.0 2147.86  4945.6 2147.50
  4954.6 2147.72  4957.1 2147.53  4962.1 2147.15  4967.8 2147.36  4977.1 2142.07
  4984.3 2131.26  4989.9 2137.23  4999.0 2124.71  5004.0 2124.71  5008.0 2123.47
  5011.2 2121.39  5011.4 2120.89  5014.9 2120.89  5015.2 2121.39  5020.6 2128.23
  5030.9 2138.90  5041.2 2145.44  5050.0 2148.98  5055.1 2149.46  5061.8 2152.81
  5070.7 2156.45  5074.5 2156.45
#Mann=5,-1,0
  4924.8    0.07       0  4934.7    0.16       0  4957.1    0.07       0
  5011.2    0.07       0  5015.2    0.07       0
Bank Sta=5011.2,5015.2
Exp/Cntr=0.3,0.1

Type RM Length L Ch R = 1,1425,18,18,18
BEGIN DESCRIPTION:
Elm 63 1424.8
END DESCRIPTION:
XS GIS Cut Line= 3
      1521290.22      6769875.27      1521345.75      6769788.50
      1521365.70      6769708.67
#Sta/Elev= 29
  4896.1 2148.29  4912.5 2148.53  4918.4 2147.34  4926.3 2147.26  4927.7 2147.24
  4933.6 2146.79  4939.7 2147.06  4948.8 2147.15  4954.8 2146.33  4964.0 2146.58
  4970.0 2145.88  4976.0 2146.68  4985.2 2140.31  4991.1 2138.32  4996.4 2123.85
  5002.0 2123.85  5007.9 2120.62  5008.2 2120.12  5011.7 2120.12  5011.9 2120.62
  5015.9 2124.09  5021.0 2127.46  5030.6 2135.02  5040.9 2147.21  5051.2 2150.09
  5057.1 2153.41  5062.3 2154.56  5079.2 2162.89  5081.4 2162.89
#Mann=5,-1,0
  4896.1    0.07       0  4926.3    0.16       0  4939.7    0.07       0
  5007.9    0.07       0  5011.9    0.07       0
Bank Sta=5007.9,5011.9
Exp/Cntr=0.3,0.1

Type RM Length L Ch R = 1,1407,30,30,30
BEGIN DESCRIPTION:
Elm 63 1406.59
END DESCRIPTION:
XS GIS Cut Line= 3
      1521285.09      6769907.43      1521363.22      6769791.32
      1521388.16      6769693.71
#Sta/Elev= 30
  4856.2 2151.65  4863.3 2150.93  4869.3 2147.87  4878.3 2148.25  4884.3 2147.02
  4899.3 2147.31  4918.7 2145.96  4921.6 2145.88  4935.3 2146.34  4956.3 2144.38
  4971.2 2144.41  4977.3 2139.38  4986.2 2128.22  4992.3 2122.76  4993.1 2118.96
  4993.4 2118.46  4997.1 2118.96  5000.4 2118.96  5009.9 2122.71  5019.3 2130.92
  5024.5 2131.67  5030.5 2140.95  5040.9 2147.96  5051.2 2150.88  5060.1 2155.23
  5065.3 2155.20  5071.8 2159.70  5082.1 2164.23  5092.1 2167.49  5096.9 2167.49
#Mann=5,-1,0
  4856.2    0.07       0  4918.7    0.16       0  4921.6    0.07       0
  4993.1    0.07       0  4997.1    0.07       0
Bank Sta=4993.1,4997.1
Exp/Cntr=0.3,0.1

Type RM Length L Ch R = 1,1377,23,23,23
BEGIN DESCRIPTION:
Elm 63 1376.81
END DESCRIPTION:
XS GIS Cut Line= 3
      1521311.15      6769913.91      1521393.60      6769791.32
      1521408.79      6769695.85
#Sta/Elev= 30
  4850.7 2146.51  4857.8 2145.99  4865.2 2146.02  4871.2 2145.17  4880.2 2145.26
  4886.2 2144.37  4901.2 2145.69  4907.2 2144.48  4922.2 2144.25  4930.1 2144.62
  4937.2 2144.33  4952.2 2138.76  4958.2 2134.60  4966.3 2127.95  4979.2 2121.94
  4988.2 2119.54  4995.4 2116.85  4995.7 2116.35  4999.2 2116.35  4999.4 2116.85
  5002.6 2116.85  5011.9 2120.44  5022.0 2130.34  5032.2 2146.54  5038.2 2148.44
  5043.3 2148.26  5062.6 2154.28  5082.8 2161.14  5091.5 2165.26  5095.1 2165.26
#Mann=3,-1,0
  4850.7    0.07       0  4995.4    0.07       0  4999.4    0.07       0
Bank Sta=4995.4,4999.4
Exp/Cntr=0.3,0.1

Type RM Length L Ch R = 1,1354,44,44,44
BEGIN DESCRIPTION:
Elm 63 1354.22
END DESCRIPTION:
XS GIS Cut Line= 3
      1521336.10      6769921.52      1521413.13      6769803.26
      1521435.54      6769711.49
#Sta/Elev= 30
  4854.1 2144.34  4870.2 2143.46  4877.9 2143.78  4883.9 2143.10  4893.0 2144.15
  4899.0 2143.24  4906.0 2143.10  4914.1 2143.62  4929.2 2143.30  4935.2 2142.51
  4941.8 2142.80  4950.3 2140.17  4956.3 2132.49  4965.5 2121.41  4971.4 2121.11
  4977.6 2116.06  4986.6 2114.37  4990.4 2113.21  4990.6 2112.71  4994.1 2112.71
  4994.4 2113.21  4995.2 2113.21  5010.9 2120.00  5020.1 2126.64  5025.3 2127.08
  5031.5 2139.18  5041.8 2147.12  5067.0 2151.67  5083.0 2157.04  5089.7 2160.38
#Mann=3,-1,0
  4854.1    0.07       0  4990.4    0.07       0  4994.4    0.07       0
Bank Sta=4990.4,4994.4
Exp/Cntr=0.3,0.1

Type RM Length L Ch R = 1,1310,44,44,44
BEGIN DESCRIPTION:
Elm 63 1309.94
END DESCRIPTION:
XS GIS Cut Line= 3
      1521352.36      6769958.43      1521448.94      6769826.04
      1521478.22      6769733.85
#Sta/Elev= 30
  4837.4 2140.35  4840.8 2140.35  4847.2 2138.98  4853.4 2134.21  4861.9 2133.14
  4868.1 2130.06  4875.1 2133.04  4882.8 2138.65  4889.0 2138.99  4897.4 2141.38
  4903.6 2140.71  4933.0 2141.37  4953.8 2139.68  4961.7 2137.77  4968.5 2131.12
  4974.7 2118.85  4987.4 2110.52  4987.6 2110.02  4991.4 2110.52  5001.3 2110.73
  5004.6 2117.24  5020.2 2129.03  5030.7 2134.63  5036.9 2143.75  5051.7 2143.94
  5062.2 2144.89  5069.1 2146.36  5074.4 2145.92  5093.2 2148.42  5098.0 2148.42
#Mann=3,-1,0
  4837.4    0.07       0  4987.4    0.07       0  4991.4    0.07       0
Bank Sta=4987.4,4991.4
Exp/Cntr=0.3,0.1

Type RM Length L Ch R = 1,1266,64,64,64
BEGIN DESCRIPTION:
Elm 63 1266.4
END DESCRIPTION:
XS GIS Cut Line= 3
      1521400.09      6769968.21      1521488.00      6769841.23
      1521509.35      6769751.58
#Sta/Elev= 30
  4842.1 2129.06  4845.3 2129.06  4854.0 2126.49  4866.7 2124.45  4874.9 2127.09
  4881.0 2125.11  4889.8 2128.84  4895.9 2126.92  4910.7 2135.05  4916.8 2131.98
  4925.6 2134.10  4931.7 2132.82  4946.5 2134.54  4952.6 2133.27  4961.4 2119.46
  4967.5 2116.05  4974.1 2108.03  4974.4 2107.53  4978.1 2108.03  4988.4 2109.47
  4995.5 2113.75  5000.8 2113.75  5005.1 2119.34  5010.2 2120.03  5020.4 2128.32
  5030.7 2139.29  5047.2 2141.34  5052.4 2140.82  5071.8 2142.42  5088.7 2145.41
#Mann=3,-1,0
  4842.1    0.07       0  4974.1    0.07       0  4978.1    0.07       0
Bank Sta=4974.1,4978.1
Exp/Cntr=0.3,0.1

Type RM Length L Ch R = 1,1202,42,42,42
BEGIN DESCRIPTION:
Elm 63 1201.71
END DESCRIPTION:
XS GIS Cut Line= 3
      1521424.01      6769971.41      1521552.02      6769844.49
      1521583.50      6769768.51
#Sta/Elev= 30
  4816.8 2126.04  4827.0 2125.66  4848.2 2121.58  4869.4 2120.61  4876.5 2122.06
  4883.6 2121.10  4890.6 2123.94  4897.7 2124.93  4904.7 2128.58  4911.8 2129.03
  4926.0 2133.02  4933.0 2127.74  4940.1 2124.22  4947.2 2112.91  4954.3 2111.52
  4959.3 2104.70  4959.6 2104.20  4963.3 2104.70  4968.4 2107.12  4975.5 2113.44
  4982.6 2109.28  4989.6 2111.94  4995.6 2109.89  5004.1 2112.50  5013.7 2116.88
  5023.6 2126.37  5032.8 2132.94  5043.0 2138.72  5058.2 2139.21  5079.3 2142.65
#Mann=5,-1,0
  4816.8    0.07       0  4959.3    0.07       0  4963.3    0.07       0
  5023.6    0.16       0  5032.8    0.07       0
Bank Sta=4959.3,4963.3
Exp/Cntr=0.3,0.1

Type RM Length L Ch R = 1,1160,37,37,37
BEGIN DESCRIPTION:
Elm 63 1159.73
END DESCRIPTION:
XS GIS Cut Line= 3
      1521465.22      6769963.84      1521585.66      6769868.36
      1521639.28      6769771.85
#Sta/Elev= 30
  4846.0 2123.22  4849.7 2121.35  4857.8 2120.29  4893.0 2117.60  4899.4 2119.88
  4907.4 2119.96  4913.8 2124.17  4921.9 2125.18  4928.3 2130.81  4935.0 2131.75
  4942.7 2128.53  4957.1 2118.06  4963.5 2110.92  4986.0 2101.08  4990.3 2100.81
  4990.6 2100.31  4994.3 2100.81  4996.1 2102.24  5002.8 2102.24  5007.2 2104.66
  5012.9 2104.58  5023.0 2108.85  5029.0 2115.41  5034.7 2113.29  5038.6 2114.97
  5045.0 2117.72  5050.7 2135.88  5068.1 2138.60  5088.4 2141.37  5110.1 2142.01
#Mann=5,-1,0
  4846.0    0.07       0  4990.3    0.07       0  4994.3    0.07       0
  5038.6    0.16       0  5068.1    0.07       0
Bank Sta=4990.3,4994.3
Exp/Cntr=0.3,0.1

Type RM Length L Ch R = 1,1123,45,45,45
BEGIN DESCRIPTION:
Elm 63 1122.57
END DESCRIPTION:
XS GIS Cut Line= 3
      1521477.19      6769973.59      1521620.38      6769883.55
      1521680.04      6769773.99
#Sta/Elev= 30
  4834.0 2124.63  4836.2 2122.42  4851.5 2122.79  4857.4 2121.14  4866.8 2120.77
  4878.7 2116.44  4888.0 2115.96  4902.3 2118.44  4909.2 2123.09  4924.5 2128.19
  4930.4 2128.79  4945.7 2127.63  4951.6 2124.20  4961.0 2121.70  4966.9 2110.01
  4973.2 2112.63  4982.2 2107.53  4988.1 2101.45  5000.9 2099.66  5001.2 2099.16
  5004.9 2099.66  5019.2 2107.93  5024.9 2107.79  5041.1 2123.79  5045.3 2126.07
  5055.0 2136.08  5084.7 2139.46  5091.2 2139.02  5106.6 2139.34  5127.9 2137.44
#Mann=5,-1,0
  4834.0    0.07       0  5000.9    0.07       0  5004.9    0.07       0
  5045.3    0.16       0  5091.2    0.07       0
Bank Sta=5000.9,5004.9
Exp/Cntr=0.3,0.1

Type RM Length L Ch R = 1,1078,56,56,56
BEGIN DESCRIPTION:
Elm 63 1077.96
END DESCRIPTION:
XS GIS Cut Line= 3
      1521482.56      6769976.87      1521659.44      6769898.74
      1521704.57      6769802.03
#Sta/Elev= 30
  4804.4 2123.86  4813.3 2123.87  4818.7 2122.79  4828.9 2123.21  4850.8 2115.59
  4859.9 2113.30  4872.7 2118.16  4883.2 2118.65  4888.6 2124.12  4905.5 2121.16
  4912.0 2121.72  4917.4 2123.58  4935.3 2123.37  4949.2 2119.55  4964.0 2105.16
  4971.1 2102.14  4985.3 2098.36  4985.6 2097.86  4989.3 2098.36  4997.8 2098.53
  5001.6 2103.08  5009.6 2108.46  5041.4 2123.95  5047.3 2123.74  5053.8 2129.99
  5064.7 2133.89  5070.2 2133.82  5093.0 2136.92  5102.3 2136.33  5104.5 2136.56
#Mann=5,-1,0
  4804.4    0.07       0  4985.3    0.07       0  4989.3    0.07       0
  5041.4    0.16       0  5102.3    0.07       0
Bank Sta=4985.3,4989.3
Exp/Cntr=0.3,0.1

Type RM Length L Ch R = 1,1022,42,42,42
BEGIN DESCRIPTION:
Elm 63 1021.67
END DESCRIPTION:
XS GIS Cut Line= 3
      1521570.46      6770063.68      1521702.84      6769936.72
      1521728.45      6769831.10
#Sta/Elev= 30
  4811.9 2132.15  4819.0 2130.51  4826.2 2131.40  4854.5 2128.01  4861.5 2125.61
  4875.6 2114.46  4882.8 2111.34  4911.1 2104.44  4918.1 2108.28  4925.3 2109.76
  4932.2 2115.11  4939.4 2116.28  4946.4 2121.20  4953.6 2122.04  4960.5 2125.11
  4967.7 2123.49  4974.7 2115.84  4981.9 2111.31  4988.8 2104.62  4993.4 2104.26
  5004.3 2097.70  5012.6 2096.63  5012.8 2096.13  5016.6 2096.63  5022.7 2097.82
  5027.9 2100.57  5061.0 2123.53  5064.5 2126.29  5076.3 2130.12  5104.0 2132.91
#Mann=4,-1,0
  4811.9    0.07       0  5012.6    0.07       0  5016.6    0.07       0
  5061.0    0.16       0
Bank Sta=5012.6,5016.6
Exp/Cntr=0.3,0.1

Type RM Length L Ch R = 1,980,34,34,34
BEGIN DESCRIPTION:
Elm 63 980.21
END DESCRIPTION:
XS GIS Cut Line= 3
      1521633.38      6770096.25      1521741.91      6769947.57
      1521786.40      6769834.70
#Sta/Elev= 30
  4809.1 2120.26  4816.7 2123.13  4822.9 2119.39  4831.4 2120.90  4837.6 2116.92
  4852.3 2116.88  4858.4 2112.86  4866.9 2111.18  4873.1 2106.07  4881.2 2104.83
  4887.8 2101.08  4894.0 2101.01  4908.7 2109.28  4917.1 2110.63  4930.7 2120.99
  4952.7 2123.29  4967.3 2121.07  4973.5 2114.35  4988.2 2107.61  4991.6 2104.37
  4995.6 2104.37  5003.5 2097.09  5015.4 2095.24  5015.7 2094.74  5019.4 2095.24
  5035.7 2098.19  5041.8 2104.19  5056.3 2110.08  5078.7 2125.71  5114.5 2133.08
#Mann=4,-1,0
  4809.1    0.07       0  5015.4    0.07       0  5019.4    0.07       0
  5056.3    0.16       0
Bank Sta=5015.4,5019.4
Exp/Cntr=0.3,0.1

Type RM Length L Ch R = 1,946,38,38,38
BEGIN DESCRIPTION:
Elm 63 946.48
END DESCRIPTION:
XS GIS Cut Line= 3
      1521657.28      6770107.07      1521772.29      6769959.51
      1521820.57      6769838.26
#Sta/Elev= 30
  4810.2 2125.18  4815.0 2123.90  4821.7 2116.84  4829.5 2111.63  4843.9 2109.93
  4858.4 2102.77  4864.8 2104.99  4879.2 2098.86  4885.6 2099.32  4893.7 2097.32
  4900.0 2098.16  4908.2 2103.51  4914.5 2102.86  4922.6 2109.16  4929.0 2110.99
  4943.5 2121.53  4949.8 2121.23  4964.3 2114.86  4972.4 2106.78  4978.7 2103.33
  4986.5 2096.38  4991.2 2094.63  4991.5 2094.13  4995.2 2094.63  5016.6 2094.97
  5031.2 2101.44  5040.9 2108.54  5052.7 2120.47  5062.0 2122.95  5127.8 2131.42
#Mann=4,-1,0
  4810.2    0.07       0  4991.2    0.07       0  4995.2    0.07       0
  5062.0    0.16       0
Bank Sta=4991.2,4995.2
Exp/Cntr=0.3,0.1

Type RM Length L Ch R = 1,908,46,46,46
BEGIN DESCRIPTION:
Elm 63 908.24
END DESCRIPTION:
XS GIS Cut Line= 3
      1521691.99      6770112.50      1521801.59      6769985.55
      1521839.14      6769871.80
#Sta/Elev= 30
  4827.4 2122.03  4846.6 2120.31  4860.7 2116.12  4874.9 2107.13  4882.6 2105.98
  4889.2 2101.24  4896.8 2099.66  4903.4 2096.93  4917.7 2096.48  4925.3 2102.42
  4939.0 2109.66  4946.2 2111.94  4952.8 2108.80  4960.5 2109.87  4967.1 2108.63
  4974.7 2104.73  4981.3 2096.06  4987.0 2093.67  4987.2 2093.17  4991.0 2093.67
  5013.6 2094.41  5025.7 2096.30  5034.7 2100.04  5045.2 2106.71  5052.2 2112.48
  5057.4 2113.18  5066.2 2117.95  5075.0 2120.96  5083.9 2123.33  5114.9 2127.73
#Mann=4,-1,0
  4827.4    0.07       0  4987.0    0.07       0  4991.0    0.07       0
  5075.0    0.16       0
Bank Sta=4987,4991
Exp/Cntr=0.3,0.1

Type RM Length L Ch R = 1,862,30,30,30
BEGIN DESCRIPTION:
Elm 63 861.95
END DESCRIPTION:
XS GIS Cut Line= 3
      1521758.16      6770121.21      1521848.24      6769990.97
      1521885.14      6769858.57
#Sta/Elev= 30
  4842.8 2117.70  4871.0 2117.42  4879.1 2107.20  4885.2 2110.58  4894.0 2101.23
  4900.1 2103.76  4907.5 2095.48  4921.0 2094.49  4935.9 2094.70  4944.0 2096.12
  4950.8 2095.73  4956.9 2093.89  4990.7 2092.48  4990.9 2091.98  4994.4 2091.98
  4994.7 2092.48  5035.4 2094.26  5042.8 2095.67  5048.0 2099.28  5056.1 2098.03
  5066.5 2099.68  5071.3 2101.35  5076.9 2103.29  5082.1 2107.30  5087.3 2118.50
  5097.7 2123.87  5116.3 2125.48  5128.8 2127.35  5136.3 2129.31  5138.6 2129.31
#Mann=4,-1,0
  4842.8    0.07       0  4990.7    0.07       0  4994.7    0.07       0
  5071.3    0.16       0
Bank Sta=4990.7,4994.7
Exp/Cntr=0.3,0.1

Type RM Length L Ch R = 1,832,74,74,74
BEGIN DESCRIPTION:
Elm 63 831.71
END DESCRIPTION:
XS GIS Cut Line= 3
      1521786.38      6770150.50      1521872.11      6770009.42
      1521915.53      6769898.71
#Sta/Elev= 30
  4831.7 2117.09  4839.6 2116.83  4846.3 2115.69  4855.0 2111.31  4860.9 2109.54
  4876.4 2112.34  4882.2 2108.83  4891.9 2107.83  4897.7 2098.30  4913.2 2093.62
  4934.5 2094.31  4955.8 2093.04  4992.7 2092.84  4994.7 2092.17  5007.1 2091.69
  5007.3 2091.19  5010.8 2091.19  5011.1 2091.69  5030.5 2093.27  5040.8 2095.06
  5046.2 2098.29  5052.0 2103.32  5062.8 2110.13  5070.6 2117.03  5076.0 2120.66
  5076.7 2120.67  5095.0 2121.49  5100.5 2122.64  5105.8 2121.92  5115.7 2122.67
#Mann=4,-1,0
  4831.7    0.07       0  5007.1    0.07       0  5011.1    0.07       0
  5076.7    0.16       0
Bank Sta=5007.1,5011.1
Exp/Cntr=0.3,0.1

Type RM Length L Ch R = 1,758,81,81,81
BEGIN DESCRIPTION:
Elm 63 757.56
END DESCRIPTION:
XS GIS Cut Line= 3
      1521843.91      6770165.65      1521924.20      6770064.76
      1521960.00      6769933.49
#Sta/Elev= 30
  4864.8 2115.43  4871.4 2115.33  4906.6 2113.42  4913.0 2113.49  4921.0 2112.61
  4926.1 2110.98  4927.4 2110.57  4935.5 2105.33  4941.8 2103.20  4949.9 2099.01
  4956.3 2098.55  4964.0 2093.94  4970.7 2092.11  5014.0 2090.29  5014.3 2089.79
  5017.8 2089.79  5018.0 2090.29  5021.5 2090.79  5031.8 2090.41  5042.2 2091.14
  5050.6 2095.82  5055.8 2096.02  5062.9 2107.15  5073.3 2111.48  5083.7 2111.83
  5095.5 2117.37  5109.5 2116.91  5114.8 2116.82  5124.9 2117.82  5129.8 2116.82
#Mann=5,-1,0
  4864.8    0.16       0  4926.1    0.07       0  5014.0    0.07       0
  5018.0    0.07       0  5109.5    0.16       0
Bank Sta=5014,5018
Exp/Cntr=0.3,0.1

Type RM Length L Ch R = 1,677,60,60,60
BEGIN DESCRIPTION:
Elm 63 676.89
END DESCRIPTION:
XS GIS Cut Line= 3
      1521979.54      6770190.58      1521996.90      6770085.37
      1522012.06      6769932.66
#Sta/Elev= 30
  4895.2 2107.42  4900.4 2107.26  4908.0 2108.03  4918.1 2108.52  4928.2 2108.51
  4948.5 2109.16  4951.0 2107.67  4956.5 2104.39  4961.6 2102.99  4968.8 2096.82
  4978.9 2092.75  4998.0 2087.92  5007.2 2087.76  5007.5 2087.26  5011.0 2087.26
  5011.2 2087.76  5019.3 2087.94  5028.8 2088.67  5033.8 2088.44  5039.4 2088.92
  5049.4 2089.06  5059.5 2088.92  5079.6 2090.61  5099.7 2100.19  5109.7 2106.68
  5116.5 2111.88  5119.8 2114.41  5129.6 2115.12  5139.9 2114.02  5155.3 2113.88
#Mann=5,-1,0
  4895.2    0.16       0  4951.0    0.07       0  5007.2    0.07       0
  5011.2    0.07       0  5116.5    0.16       0
Bank Sta=5007.2,5011.2
Exp/Cntr=0.3,0.1

Type RM Length L Ch R = 1,617,114,114,114
BEGIN DESCRIPTION:
Elm 63 616.93
END DESCRIPTION:
XS GIS Cut Line= 3
      1522028.36      6770194.99      1522056.58      6770087.54
      1522039.43      6769951.41
#Sta/Elev= 30
  4889.0 2106.24  4893.3 2106.20  4898.4 2105.17  4906.6 2105.50  4927.2 2105.57
  4938.8 2103.45  4950.2 2097.73  4958.3 2094.18  4968.6 2093.11  4974.0 2092.81
  4979.2 2090.86  4989.3 2089.64  4997.3 2087.43  5002.4 2087.43  5007.7 2086.39
  5008.0 2085.89  5011.5 2085.89  5011.7 2086.39  5019.8 2086.51  5039.9 2087.60
  5048.8 2087.59  5053.9 2088.09  5060.1 2088.02  5070.2 2090.44  5080.3 2093.88
  5100.4 2104.93  5110.5 2109.63  5120.6 2111.83  5129.2 2112.83  5137.3 2113.17
#Mann=4,-1,0
  4889.0    0.16       0  4950.2    0.07       0  5007.7    0.07       0
  5011.7    0.07       0
Bank Sta=5007.7,5011.7
Exp/Cntr=0.3,0.1

Type RM Length L Ch R = 1,503,88,88,88
BEGIN DESCRIPTION:
Elm 63 503.281
END DESCRIPTION:
XS GIS Cut Line= 3
      1522254.97      6770187.97      1522170.20      6770088.49
      1522105.00      6769938.01
#Sta/Elev= 30
  4869.3 2111.63  4872.5 2111.63  4876.4 2112.75  4879.2 2111.94  4883.0 2110.84
  4890.7 2112.74  4897.2 2108.99  4905.0 2109.14  4911.5 2100.44  4919.2 2098.38
  4925.8 2092.99  4933.5 2091.33  4947.8 2086.42  4954.4 2085.10  4980.9 2083.62
  4981.2 2083.12  4984.7 2083.12  4984.9 2083.62  5009.4 2084.14  5011.2 2084.17
  5073.7 2086.14  5087.7 2085.98  5097.1 2089.61  5102.6 2088.83  5109.5 2091.67
  5126.1 2101.13  5142.2 2102.16  5149.5 2101.34  5161.3 2106.00  5164.0 2106.00
#Mann=6,-1,0
  4869.3    0.16       0  4879.2    0.07       0  4980.9    0.07       0
  4984.9    0.07       0  5009.4    0.16       0  5011.2    0.07       0
Bank Sta=4980.9,4984.9
Exp/Cntr=0.3,0.1

Type RM Length L Ch R = 1,415,75,75,75
BEGIN DESCRIPTION:
Elm 63 4950
END DESCRIPTION:
XS GIS Cut Line= 3
      1522302.89      6770148.30      1522244.80      6770049.05
      1522132.52      6769897.64
#Sta/Elev= 30
  4885.0 2117.05  4890.9 2117.05  4912.4 2119.15  4933.9 2103.33  4949.6 2098.13
  4955.4 2093.92  4965.3 2090.42  4971.1 2086.89  4978.0 2084.27  4986.8 2082.34
  4988.5 2082.40  4992.6 2082.54  4995.7 2081.94  4996.0 2081.44  4999.5 2081.44
  4999.7 2081.94  5057.9 2083.14  5064.1 2084.20  5082.4 2084.24  5087.1 2083.85
  5093.3 2084.28  5122.6 2084.20  5128.8 2085.02  5137.2 2084.95  5150.7 2091.57
  5158.0 2097.19  5164.3 2099.12  5172.7 2103.48  5178.9 2104.38  5188.5 2104.53
#Mann=5,-1,0
  4885.0    0.07       0  4988.5    0.16       0  4995.7    0.07       0
  4999.7    0.16       0  5082.4    0.07       0
Bank Sta=4995.7,4999.7
Exp/Cntr=0.3,0.1

Type RM Length L Ch R = 1,340,69,69,69
BEGIN DESCRIPTION:
Elm 63 4949
END DESCRIPTION:
XS GIS Cut Line= 3
      1522350.64      6770126.63      1522298.98      6769996.19
      1522184.62      6769885.72
#Sta/Elev= 30
  4859.7 2115.60  4862.5 2116.18  4869.0 2111.59  4879.7 2107.62  4886.9 2103.71
  4892.2 2109.78  4911.2 2105.04  4916.6 2109.35  4922.8 2105.70  4933.5 2101.43
  4940.9 2095.94  4946.3 2097.74  4955.0 2092.08  4965.2 2087.03  4970.6 2085.41
  4976.5 2081.52  4987.3 2081.27  4993.0 2080.66  4993.2 2080.16  4996.7 2080.16
  4997.0 2080.66  5072.3 2081.57  5086.5 2082.66  5100.6 2084.80  5121.7 2094.97
  5128.9 2095.14  5135.9 2096.19  5143.1 2095.14  5150.0 2098.25  5159.0 2098.80
#Mann=3,-1,0
  4859.7    0.07       0  4993.0    0.07       0  4997.0    0.07       0
Bank Sta=4993,4997
Exp/Cntr=0.3,0.1

Type RM Length L Ch R = 1,271,61,61,61
BEGIN DESCRIPTION:
Elm 63 4947
END DESCRIPTION:
XS GIS Cut Line= 3
      1522464.55      6770112.48      1522363.32      6769977.53
      1522212.85      6769894.41
#Sta/Elev= 30
  4831.3 2113.64  4841.0 2112.31  4855.6 2105.95  4870.2 2097.07  4876.4 2097.30
  4884.8 2093.72  4891.0 2094.29  4905.6 2088.05  4911.9 2083.50  4949.3 2080.71
  4955.6 2081.86  4970.2 2079.51  4976.4 2080.15  4989.0 2079.38  4989.3 2078.88
  4993.0 2079.38  5043.8 2080.12  5066.2 2081.53  5071.9 2082.69  5087.9 2081.91
  5093.6 2086.03  5100.9 2085.19  5109.7 2082.16  5115.4 2083.53  5123.7 2082.78
  5131.5 2084.08  5137.2 2086.71  5146.6 2089.05  5158.9 2094.72  5171.9 2096.26
#Mann=3,-1,0
  4831.3    0.07       0  4989.0    0.07       0  4993.0    0.07       0
Bank Sta=4989,4993
Exp/Cntr=0.3,0.1

Type RM Length L Ch R = 1,210,47,47,47
BEGIN DESCRIPTION:
Elm 63 4946
END DESCRIPTION:
XS GIS Cut Line= 3
      1522555.68      6770017.00      1522403.12      6769932.29
      1522230.22      6769894.41
#Sta/Elev= 30
  4825.5 2100.21  4828.7 2100.21  4832.9 2096.73  4838.6 2096.34  4848.9 2092.52
  4854.6 2093.26  4870.6 2086.59  4876.3 2089.11  4892.4 2083.76  4898.1 2083.79
  4912.1 2080.81  4917.8 2077.69  4918.1 2077.19  4921.8 2077.69  4929.2 2080.30
  4941.6 2082.18  4951.9 2080.95  4957.6 2081.73  4979.3 2078.99  4999.3 2080.56
  5049.3 2079.62  5059.5 2080.86  5080.0 2087.76  5100.4 2090.64  5120.9 2091.66
  5131.2 2090.21  5136.6 2086.85  5141.7 2090.11  5151.6 2089.73  5177.0 2092.45
#Mann=3,-1,0
  4825.5    0.07       0  4917.8    0.07       0  4921.8    0.07       0
Bank Sta=4917.8,4921.8
Exp/Cntr=0.3,0.1

Type RM Length L Ch R = 1,163,114,114,114
BEGIN DESCRIPTION:
Elm 63 4945
END DESCRIPTION:
XS GIS Cut Line= 3
      1522530.05      6769913.01      1522404.43      6769884.53
      1522249.35      6769886.80
#Sta/Elev= 30
  4871.2 2088.21  4876.4 2090.31  4886.6 2088.10  4896.9 2083.64  4907.1 2078.00
  4914.4 2074.99  4919.5 2074.37  4925.6 2073.26  4925.9 2072.76  4929.4 2072.76
  4929.6 2073.26  4937.9 2073.47  4962.6 2073.58  4968.7 2073.45  5002.2 2073.30
  5009.4 2073.90  5019.4 2077.43  5029.4 2081.72  5039.4 2082.15  5049.4 2080.12
  5059.4 2075.33  5079.4 2080.35  5089.4 2081.69  5099.4 2084.95  5109.4 2087.26
  5119.4 2088.88  5129.4 2089.72  5139.4 2090.71  5149.4 2091.52  5155.1 2093.02
#Mann=3,-1,0
  4871.2    0.07       0  4925.6    0.07       0  4929.6    0.07       0
Bank Sta=4925.6,4929.6
Exp/Cntr=0.3,0.1

Type RM Length L Ch R = 1,49,0,0,0
BEGIN DESCRIPTION:
Elm 63 4944
END DESCRIPTION:
XS GIS Cut Line= 3
      1522530.04      6769863.02      1522358.65      6769786.49
      1522258.99      6769842.46
#Sta/Elev= 30
  4812.3 2093.61  4817.8 2090.18  4828.8 2087.25  4835.6 2086.19  4841.0 2088.81
  4858.8 2080.35  4864.3 2080.21  4872.6 2076.48  4882.0 2074.23  4894.5 2073.30
  4927.3 2073.50  4933.9 2074.35  4939.4 2079.30  4949.2 2081.65  4957.1 2080.90
  4962.6 2077.36  4971.1 2074.16  4983.8 2071.45  4984.1 2070.95  4987.8 2071.45
  5011.6 2073.07  5017.3 2075.38  5027.1 2075.66  5033.3 2077.03  5039.0 2082.17
  5049.2 2084.87  5055.0 2088.12  5061.5 2089.40  5092.6 2088.80  5114.3 2090.92
#Mann=3,-1,0
  4812.3    0.07       0  4983.8    0.07       0  4987.8    0.07       0
Bank Sta=4983.8,4987.8
Exp/Cntr=0.3,0.1

Chan Stop Cuts=-1
