--- Elm 74.prj (project) ---

Proj Title=Elm 74 Base Level Engineering
Current Plan=p01
Default Exp/Contr=0.3,0.1
English Units
Geom File=g01
Flow File=f01
Plan File=p01
Y Axis Title=Elevation
X Axis Title(PF)=Main Channel Distance
X Axis Title(XS)=Station
BEGIN DESCRIPTION:
Elm 74
END DESCRIPTION:
DSS Export Rating Curves= 0
DSS Export Rating Curve Sorted= 0
DSS Export Volume Flow Curves= 0
DXF OffsetX= 0
DXF OffsetY= 0
DXF ScaleX= 1
DXF ScaleY= 10

--- Elm 74.p01 (plan) ---

Plan Title=Multiple Run
Short Identifier=Multiple
Geom File=g01
Flow File=f01
Subcritical Flow
K Sum by GR= 0
Std Step Tol= 0.01
Critical Tol= 0.01
Num of Std Step Trials= 20
Max Error Tol= 0.3
Flow Tol Ratio= 0.001
Split Flow NTrial= 30
Split Flow Tol= 0.02
Split Flow Ratio= 0.02
Log Output Level= 0
Friction Slope Method= 1
Unsteady Friction Slope Method= 2
Unsteady Bridges Friction Slope Method= 1
Parabolic Critical Depth
Global Vel Dist=  1 , 1 , 1
Global Log Level= 0
CheckData=True
Encroach Param= -1, 0, 0, 0
BEGIN DESCRIPTION:
Multiple Run
END DESCRIPTION:

--- Elm 74.f01 (steady flow) ---

Flow Title=Multiple
Number of Profiles=7
Profile Names=10-year,25-year,50-year,1pct_min,100-year,1pct_plu,500-year
River Rch & RM= Elm 74,Reach-1,19784
     351     505     639     502     804    1110    1290
River Rch & RM= Elm 74,Reach-1,13957
     418     605     767     603     967    1330    1560
River Rch & RM= Elm 74,Reach-1,9437
     699    1040    1340    1070    1720    2360    2860
River Rch & RM= Elm 74,Reach-1,6663
     686    1010    1300    1030    1660    2280    2730
Boundary for River Rch & Prof#=Elm 74,Reach-1,1
Up Type=0
Dn Type=3
Dn Slope=0.005
Boundary for River Rch & Prof#=Elm 74,Reach-1,2
Up Type=0
Dn Type=3
Dn Slope=0.005
Boundary for River Rch & Prof#=Elm 74,Reach-1,3
Up Type=0
Dn Type=3
Dn Slope=0.005
Boundary for River Rch & Prof#=Elm 74,Reach-1,4
Up Type=0
Dn Type=3
Dn Slope=0.005
Boundary for River Rch & Prof#=Elm 74,Reach-1,5
Up Type=0
Dn Type=3
Dn Slope=0.005
Boundary for River Rch & Prof#=Elm 74,Reach-1,6
Up Type=0
Dn Type=3
Dn Slope=0.005
Boundary for River Rch & Prof#=Elm 74,Reach-1,7
Up Type=0
Dn Type=3
Dn Slope=0.005

--- Elm 74.g01 (geometry) ---

Geom Title=Existing Conditions
Program Version=4.10

River Reach=Elm 74          ,Reach-1
Reach XY= 30
        1524455.        6760088.      1524956.33      6760584.68
      1525170.36      6760387.89      1525415.45      6760586.97
      1525849.07      6760490.25      1526725.65       6761157.4
      1526910.46      6762290.45      1527838.55      6763220.86
      1527862.69      6763644.47      1528406.63      6764184.88
      1528894.46      6763989.08      1529580.03      6764388.51
      1530094.67      6764088.87      1530694.03      6764427.62
      1530660.45      6764641.01        1530855.        6764638.
      1531148.03      6765188.25      1530760.05      6765390.28
      1531553.46      6765893.85        1531355.        6766388.
       1531805.4      6766658.13      1531557.99      6767086.54
      1531894.22       6767277.8      1531810.36       6767590.7
      1532347.51      6768081.31      1532458.83      6768736.42
      1533151.46      6769739.46      1533008.75      6770736.45
      1533291.69       6771174.6        1533655.        6771288.

Type RM Length L Ch R = 1 ,19784   ,115,115,115
BEGIN DESCRIPTION:
Elm 74 4328
END DESCRIPTION:
XS GIS Cut Line= 3
      1524447.39      6760287.45      1524553.33      6760142.04
      1524646.32      6760032.23
#Sta/Elev= 30
  4820.1 2270.26  4825.1 2270.96  4831.8 2268.99  4839.7 2267.55  4845.9 2268.04
  4868.9 2267.08  4881.5 2264.59  4931.7 2261.51    4961 2261.44  4990.4  2262.2
  4996.6  2261.1  5005.2 2260.99  5016.4 2255.77  5016.7 2255.27  5020.2 2255.27
  5020.4 2255.77  5031.9  2256.6  5039.7 2262.02  5046.2 2264.53    5054 2269.61
  5068.2 2274.81  5074.8 2275.09  5082.5 2276.82  5089.1 2276.86  5096.8 2278.06
  5110.1 2278.47  5117.7 2279.52  5124.2 2279.12  5138.5 2280.09  5143.9 2281.12
#Mann= 3 ,-1 , 0
  4820.1     .16       0  5016.4     .07       0  5020.4     .16       0
Bank Sta=5016.4,5020.4
XS Rating Curve= 0 ,0
Exp/Cntr=0.3,0.1

Type RM Length L Ch R = 1 ,19669   ,133,133,133
BEGIN DESCRIPTION:
Elm 74 4326
END DESCRIPTION:
XS GIS Cut Line= 3
      1524521.15      6760387.31      1524653.37      6760191.95
      1524744.71      6760102.99
#Sta/Elev= 30
  4764.1 2271.91  4774.6 2271.68  4780.6 2270.72  4795.6 2269.88  4801.6  2268.6
  4810.6 2268.03  4837.6 2264.27  4846.5 2264.25  4873.5 2262.19  4888.5 2261.88
  4909.5 2260.24  4918.4  2260.2  4954.4 2257.24  4960.4 2256.26  4975.4 2256.31
  4988.3 2253.59  4988.6 2253.09  4992.1 2253.09  4992.3 2253.59  4999.4  2255.1
    5011 2255.31  5039.3 2258.31  5046.3 2258.59  5067.6 2262.64  5074.6 2265.45
  5081.8 2266.77  5095.9 2272.39  5102.9 2272.93  5110.1    2275  5127.5 2276.84
#Mann= 3 ,-1 , 0
  4764.1     .16       0  4988.3     .07       0  4992.3     .16       0
Bank Sta=4988.3,4992.3
XS Rating Curve= 0 ,0
Exp/Cntr=0.3,0.1

Type RM Length L Ch R = 1 ,19536   ,122,122,122
BEGIN DESCRIPTION:
Elm 74 4325
END DESCRIPTION:
XS GIS Cut Line= 3
      1524605.79      6760474.12      1524749.63       6760282.5
      1524837.16       6760182.1
#Sta/Elev= 30
  4760.4 2266.07  4770.9 2265.21  4779.2 2266.38  4793.1 2265.61    4800 2264.65
  4820.9  2264.1  4835.4 2262.75  4843.1 2262.53    4850 2261.01  4870.8 2259.34
  4879.2 2259.47  4885.4 2258.41  4906.3 2257.51  4956.3 2256.18  4970.8 2256.86
  4985.4 2256.67  4993.1  2255.5  4997.7 2250.03  4997.9 2249.53  5001.4 2249.53
  5001.7 2250.03  5020.8 2252.48  5035.1 2254.97  5042.7 2259.53  5063.6 2266.77
  5071.2 2268.99  5077.8 2270.29  5085.4 2272.68  5098.8  2275.2  5133.2 2278.52
#Mann= 3 ,-1 , 0
  4760.4     .16       0  4997.7     .07       0  5001.7     .16       0
Bank Sta=4997.7,5001.7
XS Rating Curve= 0 ,0
Exp/Cntr=0.3,0.1

Type RM Length L Ch R = 1 ,19414   ,105,105,105
BEGIN DESCRIPTION:
Elm 74 19406.227
END DESCRIPTION:
XS GIS Cut Line= 3
      1524717.26      6760552.28      1524842.08      6760359.62
      1524924.78      6760224.59
#Sta/Elev= 30
  4781.9 2269.24  4798.9 2268.67  4841.4 2262.25  4898.7  2256.7  4906.1  2254.5
  4913.9 2255.84    4929 2255.08    4935 2253.75  4950.2    2254  4965.3 2252.03
  4977.6 2252.33  4986.4 2253.65  5001.5 2253.16  5007.5 2252.22  5009.5 2249.92
  5015.3 2249.92  5020.9 2248.69  5021.2 2248.19  5024.9 2248.69  5028.8 2250.25
  5036.8 2256.08  5086.8 2263.97  5102.3 2269.88  5108.1 2269.53  5117.7 2271.75
  5123.6 2271.37    5139 2273.76  5144.9 2273.27  5160.3  2274.5  5169.8 2273.83
#Mann= 3 ,-1 , 0
  4781.9     .16       0  5020.9     .07       0  5024.9     .16       0
Bank Sta=5020.9,5024.9
XS Rating Curve= 0 ,0
Exp/Cntr=0.3,0.1

Type RM Length L Ch R = 1 ,19309   ,154,154,154
BEGIN DESCRIPTION:
Elm 74 19309.29
END DESCRIPTION:
XS GIS Cut Line= 3
      1524807.59      6760597.85      1524913.95      6760430.71
      1524954.98      6760262.25
#Sta/Elev= 30
  4821.9 2269.93  4824.2 2269.93    4827 2267.78  4835.3 2267.37  4842.3 2266.44
  4848.2  2264.1  4857.3 2263.96  4899.8 2257.95  4915.1 2254.66    4921 2251.05
  4942.2 2249.67  4951.5 2250.41  4957.4 2248.55  4972.6 2249.19  4997.7 2246.53
    4998 2246.03  5001.7 2246.53  5018.7 2252.16  5047.1 2253.07  5083.6 2256.11
  5088.8 2255.96  5094.8 2257.66  5115.4 2259.56  5130.5 2260.09    5136 2261.54
  5166.9 2263.81  5172.2 2266.26  5177.3 2264.68  5187.5 2266.14  5193.4 2267.86
#Mann= 4 ,-1 , 0
  4821.9     .07       0  4835.3     .16       0  4997.7     .07       0
  5001.7     .16       0
Bank Sta=4997.7,5001.7
XS Rating Curve= 0 ,0
Exp/Cntr=0.3,0.1

Type RM Length L Ch R = 1 ,19155   ,77,77,77
BEGIN DESCRIPTION:
Elm 74 19155.39
END DESCRIPTION:
XS GIS Cut Line= 3
      1524913.95      6760675.94      1524953.01       6760591.3
      1524959.52       6760326.5
#Sta/Elev= 30
  4897.7 2275.74  4906.4 2274.59  4912.1 2272.95  4917.6 2272.16  4928.5 2269.72
  4940.5  2265.9  4950.5 2264.84  4957.9 2264.33  4963.4 2264.28  4972.5  2262.6
  4980.9 2260.54  4986.4 2245.94    4988 2244.89  4988.2 2244.39  4991.7 2244.39
    4992 2244.89  4995.1 2244.89  5004.2 2246.58  5014.2 2247.67  5044.2 2248.13
  5084.3  2249.7  5124.3 2249.73  5154.3 2251.08  5184.3  2253.6  5194.3 2254.95
  5214.3 2256.95  5224.3 2258.27  5244.3 2259.42  5252.5 2260.41  5255.8 2260.41
#Mann= 3 ,-1 , 0
  4897.7     .16       0    4988     .07       0    4992     .16       0
Bank Sta=4988,4992
XS Rating Curve= 0 ,0
Exp/Cntr=0.3,0.1

Type RM Length L Ch R = 1 ,19078   ,114,114,114
BEGIN DESCRIPTION:
Elm 74 19078.37
END DESCRIPTION:
XS GIS Cut Line= 3
       1525033.3      6760699.78      1525028.96      6760586.96
      1524987.73      6760346.06
#Sta/Elev= 30
  4888.5 2269.05  4891.9 2269.05  4900.3 2267.12  4920.3  2266.4  4930.3 2264.68
  4974.9    2259  4980.3 2256.36  4990.4 2252.77  4998.4 2247.94  5003.4 2247.94
  5010.5 2243.64  5018.6 2242.48  5018.9 2241.98  5022.4 2241.98  5022.6 2242.48
  5030.3 2244.93  5040.9 2245.83  5050.3 2245.32  5055.3 2245.95  5061.2 2245.29
  5071.4 2245.17  5081.5 2245.81  5101.8 2246.01  5132.2 2249.38  5162.7 2250.72
  5170.4 2251.88  5203.3 2254.29  5223.5 2256.22  5242.3 2259.02  5245.8 2259.02
#Mann= 4 ,-1 , 0
  4888.5     .07       0  5018.6     .07       0  5022.6     .07       0
  5030.3     .16       0
#XS Ineff= 2 , 0
       0                    5040       0    2255
Permanent Ineff=
       F       F
Bank Sta=5018.6,5022.6
XS Rating Curve= 0 ,0
Exp/Cntr=0.3,0.1

Type RM Length L Ch R = 1 ,18964   ,93,93,93
BEGIN DESCRIPTION:
Elm 74 18964.3
END DESCRIPTION:
XS GIS Cut Line= 3
       1525122.3      6760686.84      1525059.35      6760493.65
      1525020.33      6760302.88
#Sta/Elev= 30
  4795.2 2265.06  4838.1    2263  4864.8 2260.47    4870 2260.94  4888.6 2258.53
  4896.7 2256.43  4901.9 2256.38  4928.5 2251.38  4933.8 2252.28  4941.2 2249.83
  4951.7 2243.13  4960.5 2243.33  4972.8 2241.46  4983.3  2241.6  4992.4 2242.81
  4997.3 2241.45  5004.1 2240.78  5040.5 2240.38  5040.7 2239.88  5044.2 2239.88
  5044.5 2240.38  5055.2 2245.96  5065.4 2249.67  5085.8 2252.71  5092.9 2254.81
    5098  2254.8  5126.6 2259.02  5143.4 2260.01  5148.5 2259.03  5193.1 2261.25
#Mann= 4 ,-1 , 0
  4795.2     .07       0  4928.5     .16       0  5040.5     .07       0
  5044.5     .16       0
Bank Sta=5040.5,5044.5
XS Rating Curve= 0 ,0
Exp/Cntr=0.3,0.1

Type RM Length L Ch R = 1 ,18871   ,86,86,86
BEGIN DESCRIPTION:
Elm 74 18870.8
END DESCRIPTION:
XS GIS Cut Line= 3
      1525124.45      6760688.97      1525122.28      6760426.37
      1525009.69      6760225.01
#Sta/Elev= 30
    4733 2265.06    4804  2260.4    4844 2252.95  4860.7 2250.87    4884 2247.62
    4914  2245.4  4995.6 2242.41  4997.9 2239.13  4998.1 2238.63  5001.9 2239.13
  5015.8  2240.7  5021.6 2243.05  5028.1 2248.79  5037.5  2254.5  5059.2 2260.61
  5096.9 2262.29  5102.7 2263.71  5108.4 2262.47  5118.6    2265  5124.4 2263.39
  5140.3 2267.35  5146.1 2264.82    5162 2268.65  5167.8 2265.71  5183.7 2268.46
  5189.5  2265.2  5199.7 2267.17  5205.4 2264.28  5221.4 2267.09  5226.3 2265.19
#Mann= 4 ,-1 , 0
    4733     .07       0  4860.7     .16       0  4997.9     .07       0
  5001.9     .16       0
Bank Sta=4997.9,5001.9
XS Rating Curve= 0 ,0
Exp/Cntr=0.3,0.1

Type RM Length L Ch R = 1 ,18785   ,291,291,291
BEGIN DESCRIPTION:
Elm 74 18784.75
END DESCRIPTION:
XS GIS Cut Line= 3
      1525172.19      6760699.81       1525193.9      6760391.65
       1525193.9      6760285.28
#Sta/Elev= 30
  4688.7    2266  4692.1    2266  4700.5 2265.01  4730.6 2262.92  4770.7 2259.56
  4790.8 2256.21  4797.8 2253.69  4802.8 2252.68  4810.8 2249.48  4820.8 2247.15
    4826 2246.69    4881 2244.26  4911.1 2243.45  4921.1 2242.36  4931.1 2242.02
  4944.2 2240.65  4951.2 2240.89  4981.2 2240.63  4991.3 2239.97    4997 2238.17
    5002 2238.17  5009.3 2236.77  5009.5 2236.27    5013 2236.27  5013.3 2236.77
  5021.3 2242.32  5041.3 2259.95  5071.3 2263.99  5100.1 2271.07    5104 2271.07
#Mann= 4 ,-1 , 0
  4688.7     .07       0    4826     .16       0  5009.3     .07       0
  5013.3     .16       0
Bank Sta=5009.3,5013.3
XS Rating Curve= 0 ,0
Exp/Cntr=0.3,0.1

Type RM Length L Ch R = 1 ,18494   ,77,77,77
BEGIN DESCRIPTION:
Elm 74 18494.42
END DESCRIPTION:
XS GIS Cut Line= 3
      1525337.13      6760730.18      1525406.57      6760584.79
      1525326.26      6760278.77
#Sta/Elev= 30
  4837.9 2264.62    4880 2262.68  4906.8 2262.22  4918.8 2260.69    4929 2253.96
  4935.9  2248.5  4941.5 2248.09  4958.6 2239.67  4964.2 2238.64  4973.3 2233.73
  4979.3 2229.17  4979.6 2228.67  4983.1 2228.67  4983.3 2229.17  4986.8 2229.41
  4994.5 2231.64    4999 2231.64    5006 2233.09  5016.4 2233.99  5047.4  2234.4
  5068.8 2235.47  5078.4 2237.22  5171.5 2242.99  5192.1 2245.56  5202.5 2245.06
  5219.9 2246.28  5254.2 2250.27  5285.2 2258.62  5305.9 2261.43  5315.4 2261.34
#Mann= 4 ,-1 , 0
  4837.9     .07       0    4880     .16       0  4979.3     .07       0
  4983.3     .16       0
Bank Sta=4979.3,4983.3
XS Rating Curve= 0 ,0
Exp/Cntr=0.3,0.1

Type RM Length L Ch R = 1 ,18417   ,152,152,152
BEGIN DESCRIPTION:
Elm 74 18417.49
END DESCRIPTION:
XS GIS Cut Line= 3
       1525491.2      6760728.03      1525482.52      6760584.79
      1525359.65      6760214.02
#Sta/Elev= 30
  4859.7  2256.8  4877.2 2256.68  4882.2 2257.68  4925.5  2255.1  4939.9 2252.52
  4953.7  2245.7  4969.9 2238.05    4980 2234.53  4999.1 2229.51  5003.2 2229.51
  5006.2 2228.09  5006.4 2227.59  5010.2 2228.09  5013.4  2228.5  5020.9 2231.63
  5031.4 2232.45  5071.6  2232.8  5103.2 2234.68  5115.7 2236.41  5134.9 2236.69
  5140.2 2237.73  5157.8 2238.93  5210.5 2240.68    5267 2244.05  5284.3 2246.36
  5305.3 2253.68  5325.1 2259.63  5356.8 2263.99  5368.5 2267.66  5393.8 2271.83
#Mann= 5 ,-1 , 0
  4859.7     .16       0  4925.5     .07       0  4953.7     .16       0
  5006.2     .07       0  5010.2     .16       0
Bank Sta=5006.2,5010.2
XS Rating Curve= 0 ,0
Exp/Cntr=0.3,0.1

Type RM Length L Ch R = 1 ,18265   ,115,115,115
BEGIN DESCRIPTION:
Elm 74 18265.23
END DESCRIPTION:
XS GIS Cut Line= 3
      1525595.37       6760643.4      1525556.31      6760497.99
      1525482.79      6760232.03
#Sta/Elev= 30
    4851 2243.08  4871.9 2246.26  4887.7 2244.88    4898 2241.85  4911.9 2233.07
  4918.7 2227.19    4936 2219.48  4949.9 2214.42  4950.1 2213.92  4953.9 2214.42
  4970.5 2217.41  4986.7 2218.12  4991.9 2221.93  5004.2 2222.02  5021.2 2218.47
  5026.4 2222.67  5043.1 2225.47  5053.4 2225.25  5060.7 2220.17  5074.2 2227.99
  5084.6 2231.63  5146.8 2239.79  5188.3 2243.15  5198.7 2245.06  5208.4 2249.67
  5213.6 2249.03  5219.4 2253.44  5240.2  2260.1  5253.1 2259.54  5277.5 2261.14
#Mann= 4 ,-1 , 0
    4851     .07       0    4936     .16       0  4949.9     .07       0
  4953.9     .16       0
Bank Sta=4949.9,4953.9
XS Rating Curve= 0 ,0
Exp/Cntr=0.3,0.1

Type RM Length L Ch R = 1 ,18150   ,119,119,119
BEGIN DESCRIPTION:
Elm 74 18150.08
END DESCRIPTION:
XS GIS Cut Line= 3
      1525619.24      6760643.38      1525643.11       6760445.9
      1525623.67      6760262.24
#Sta/Elev= 30
  4794.3 2238.49  4797.6 2238.71  4802.7 2235.73    4840 2238.66  4860.2 2239.55
  4884.6 2237.94  4890.4 2236.82  4928.8 2233.09  4940.7 2231.69  4960.9 2227.42
  4966.6 2224.23  4971.6 2223.25    4981 2217.26  4987.6 2209.61  4987.9 2209.11
  4991.4 2209.11  4991.6 2209.61  5001.2 2211.26  5019.5 2222.14  5024.5 2221.84
  5031.3 2226.17  5041.4 2231.58  5061.5 2239.52  5071.6 2241.12  5081.6 2244.83
  5101.7 2257.06  5117.3 2265.43  5122.3 2264.08    5152 2271.89  5177.9 2275.13
#Mann= 4 ,-1 , 0
  4794.3     .07       0  4928.8     .16       0  4987.6     .07       0
  4991.6     .16       0
Bank Sta=4987.6,4991.6
XS Rating Curve= 0 ,0
Exp/Cntr=0.3,0.1

Type RM Length L Ch R = 1 ,18031   ,104,104,104
BEGIN DESCRIPTION:
Elm 74 18031.25
END DESCRIPTION:
XS GIS Cut Line= 4
      1525636.59      6760608.68      1525745.11      6760491.48
      1525764.64      6760320.04      1525768.98        6760268.
#Sta/Elev= 30
  4836.3 2234.95  4838.8 2234.95  4842.7 2231.22    4850 2232.86  4856.9  2229.1
  4864.2 2232.29    4871 2228.84  4885.2 2234.31    4892 2232.71  4899.4  2234.1
  4906.2 2232.91  4927.7 2232.64  4962.9  2228.8  4970.2 2227.43  4985.9 2221.72
  4991.2 2220.22    4995 2214.21  5000.3 2214.21  5009.6 2209.03  5017.7 2208.18
  5017.9 2207.68  5021.7 2208.18  5029.7 2213.33    5037 2220.63  5059.9 2230.18
  5090.1 2246.07  5126.5 2260.56  5172.1 2267.14  5190.7 2271.12  5220.8 2273.99
#Mann= 4 ,-1 , 0
  4836.3     .07       0  4985.9     .16       0  5017.7     .07       0
  5021.7     .16       0
Bank Sta=5017.7,5021.7
XS Rating Curve= 0 ,0
Exp/Cntr=0.3,0.1

Type RM Length L Ch R = 1 ,17927   ,56,56,56
BEGIN DESCRIPTION:
Elm 74 17926.84
END DESCRIPTION:
XS GIS Cut Line= 3
      1525758.15      6760691.09      1525851.45      6760487.14
       1525825.4       6760298.3
#Sta/Elev= 30
  4779.6 2240.56  4826.8 2238.43    4838 2236.66    4849 2236.31  4860.8 2233.27
  4883.8  2229.4  4906.9 2226.92  4924.4 2226.83  4940.6 2224.72  4952.9 2223.22
  4958.9 2215.88  4969.9 2208.42  4973.9 2204.86  4974.2 2204.36  4977.9 2204.86
  4991.9  2210.2  4998.9 2215.68  5002.1 2217.04    5006 2217.04  5011.3  2222.3
  5016.3 2221.55  5023.2 2225.98  5043.4 2235.02  5073.7 2243.61  5083.2 2246.13
  5088.2 2246.05  5093.9 2248.93  5124.1 2255.89  5165.2 2260.97  5194.5 2262.95
#Mann= 4 ,-1 , 0
  4779.6     .07       0  4940.6     .16       0  4973.9     .07       0
  4977.9     .16       0
Bank Sta=4973.9,4977.9
XS Rating Curve= 0 ,0
Exp/Cntr=0.3,0.1

Type RM Length L Ch R = 1 ,17871   ,79,79,79
BEGIN DESCRIPTION:
Elm 74 17870.64
END DESCRIPTION:
XS GIS Cut Line= 3
      1525771.16        6760715.      1525894.85      6760532.71
      1525879.72      6760281.96
#Sta/Elev= 30
  4771.5 2241.12  4837.5 2237.84  4858.5 2237.54  4879.5 2234.31  4888.4 2231.86
  4894.4  2231.7  4900.8 2229.44  4909.4 2227.69  4915.4 2227.62  4924.3 2225.34
  4937.1 2223.72  4948.4 2223.35  4960.3 2223.87  4973.3 2216.27  4981.3  2208.4
  4987.3 2206.34  4989.6 2204.13  4989.9 2203.63  4993.6 2204.13  4996.7 2204.13
  5026.6 2218.27  5046.6    2224  5066.6 2226.46    5072 2229.53  5156.8 2249.86
  5166.8 2251.31  5186.9 2252.49  5235.1 2253.26  5240.1 2256.25    5243  2256.4
#Mann= 4 ,-1 , 0
  4771.5     .07       0  4948.4     .16       0  4989.6     .07       0
  4993.6     .16       0
Bank Sta=4989.6,4993.6
XS Rating Curve= 0 ,0
Exp/Cntr=0.3,0.1

Type RM Length L Ch R = 1 ,17792   ,66,66,66
BEGIN DESCRIPTION:
Elm 74 17792.01
END DESCRIPTION:
XS GIS Cut Line= 3
      1525829.72      6760751.93      1525966.46      6760556.58
       1525938.4      6760241.38
#Sta/Elev= 30
  4756.5 2241.03  4857.2 2235.98  4878.2 2232.46  4884.3 2233.07    4893 2230.64
  4899.1 2232.28  4913.9 2225.83  4934.8 2220.26  4943.5 2219.48  4964.5  2214.2
  4970.6 2214.28  4985.4 2207.23    4989 2202.69  4989.3 2202.19    4993 2202.69
  5003.6 2203.21  5023.6 2212.99  5033.7 2215.65  5073.8 2222.04    5124 2227.85
  5164.2 2237.36  5179.9 2237.56  5184.9 2239.82  5194.3 2240.28  5224.4 2239.12
  5254.6  2241.4  5284.7 2239.95  5291.5 2240.03  5296.5 2242.21  5311.4 2241.45
#Mann= 3 ,-1 , 0
  4756.5     .16       0    4989     .07       0    4993     .16       0
Bank Sta=4989,4993
XS Rating Curve= 0 ,0
Exp/Cntr=0.3,0.1

Type RM Length L Ch R = 1 ,17726   ,54,54,54
BEGIN DESCRIPTION:
Elm 74 17725.52
END DESCRIPTION:
XS GIS Cut Line= 3
      1525853.64      6760767.06      1526014.21      6760597.81
      1525999.08      6760241.33
#Sta/Elev= 30
  4766.1 2240.44  4794.6 2239.63  4808.7 2238.13  4872.6 2235.53  4907.8 2233.07
  4915.1 2228.55    4922 2227.95  4936.1 2220.71  4950.3 2215.55  4978.6 2214.69
  4992.8 2205.57  4996.3 2202.26  5001.8 2202.26  5007.2 2200.34  5007.5 2199.84
  5011.2 2200.34  5019.2 2202.38  5039.2 2205.48  5059.3 2215.34  5069.3 2222.95
  5101.5 2222.04  5109.3 2223.08  5129.3 2223.53  5139.3 2224.53  5169.4 2230.74
  5179.4 2230.51  5199.4 2225.57  5209.4 2224.88  5259.4 2228.16  5356.2 2232.98
#Mann= 3 ,-1 , 0
  4766.1     .16       0  5007.2     .07       0  5011.2     .16       0
Bank Sta=5007.2,5011.2
XS Rating Curve= 0 ,0
Exp/Cntr=0.3,0.1

Type RM Length L Ch R = 1 ,17672   ,74,74,74
BEGIN DESCRIPTION:
Elm 74 17671.89
END DESCRIPTION:
XS GIS Cut Line= 3
      1525877.48       6760773.6      1526055.44      6760632.54
      1526268.15      6760419.83
#Sta/Elev= 30
  4777.5 2239.62  4901.4 2234.48  4914.7 2232.76  4922.2 2231.06  4928.6 2227.17
  4936.6 2225.26  4957.5 2214.18  4965.5 2210.43  4971.9 2209.23  4978.5  2205.4
  4986.3 2203.03  5000.7    2201  5007.8 2201.29  5021.6 2198.89  5026.7 2196.71
  5026.9 2196.21  5030.7 2196.71  5064.1 2201.23  5071.1 2199.88  5085.3 2200.19
  5092.3 2203.05  5106.5 2212.34  5113.6 2215.12  5148.9 2219.46  5191.3 2231.45
  5198.4 2230.91  5205.5  2233.6  5233.8 2238.83    5255 2240.69  5305.4 2251.53
#Mann= 3 ,-1 , 0
  4777.5     .16       0  5026.7     .07       0  5030.7     .16       0
Bank Sta=5026.7,5030.7
XS Rating Curve= 0 ,0
Exp/Cntr=0.3,0.1

Type RM Length L Ch R = 1 ,17598   ,111,111,111
BEGIN DESCRIPTION:
Elm 74 17597.52
END DESCRIPTION:
XS GIS Cut Line= 3
      1525888.37       6760808.3      1526111.86      6760684.62
      1526318.06      6760519.66
#Sta/Elev= 30
  4757.3 2240.36  4799.2 2236.99    4916 2233.73    4932 2232.12  4947.7 2226.49
  4953.8 2219.62  4975.5 2206.64    4982 2201.58  4991.6 2197.33  4997.3 2197.01
  5002.9 2194.88  5003.1 2194.38  5006.9 2194.88  5019.2 2196.63  5027.2 2202.37
  5041.7 2210.58  5055.2 2212.09  5076.9 2212.13  5112.1 2214.33  5119.2 2217.46
  5132.9 2221.58  5161.7 2228.18  5176.1 2230.49  5190.5  2230.6  5196.9 2232.77
  5204.9 2232.55  5211.3 2234.65  5219.3 2233.79    5269 2241.35  5276.8 2241.43
#Mann= 3 ,-1 , 0
  4757.3     .16       0  5002.9     .07       0  5006.9     .16       0
Bank Sta=5002.9,5006.9
XS Rating Curve= 0 ,0
Exp/Cntr=0.3,0.1

Type RM Length L Ch R = 1 ,17487   ,118,118,118
BEGIN DESCRIPTION:
Elm 74 17486.72
END DESCRIPTION:
XS GIS Cut Line= 3
      1525916.59      6760918.97       1526153.1      6760782.28
      1526378.13      6760572.38
#Sta/Elev= 30
  4727.1 2248.12  4858.5 2233.97  4864.3  2230.3  4874.3 2231.01  4880.1 2226.74
  4895.8 2227.97  4901.6 2223.87  4917.4 2222.48  4923.1 2217.52  4929.7 2217.45
  4933.1 2217.41  4938.9 2212.82  4954.7 2210.26  4960.5 2203.86  4988.9 2193.44
  4989.2 2192.94  4992.9 2193.44  4994.2 2193.84  5032.8 2199.63  5040.1  2198.2
    5047 2201.05  5054.3 2197.42  5075.3 2207.55  5089.5  2208.7  5096.8 2206.73
  5103.6 2209.82  5125.1  2210.4  5188.6 2229.83    5238 2232.41    5308 2247.52
#Mann= 5 ,-1 , 0
  4727.1     .16       0  4929.7     .07       0  4988.9     .07       0
  4992.9     .07       0  4994.2     .16       0
Bank Sta=4988.9,4992.9
XS Rating Curve= 0 ,0
Exp/Cntr=0.3,0.1

Type RM Length L Ch R = 1 ,17369   ,72,72,72
BEGIN DESCRIPTION:
Elm 74 17368.62
END DESCRIPTION:
XS GIS Cut Line= 3
      1526064.08      6760942.89      1526265.94      6760801.81
      1526448.25      6760595.63
#Sta/Elev= 30
  4752.3 2241.42  4814.4 2234.31  4842.2  2227.4  4850.9 2226.98  4873.3 2220.58
  4886.6 2217.25  4892.7  2211.3  4907.6 2208.66  4913.7 2201.83  4922.4 2202.74
  4928.5 2196.92  4943.3 2206.12  4949.4 2201.78  4958.2 2206.13  4964.3  2202.4
    4973 2202.32  4979.1 2198.44  4985.2 2198.22  4997.5 2194.49  5021.7 2193.86
  5029.3 2190.47  5041.5 2187.86  5041.8 2187.36  5045.5 2187.86  5050.2 2188.03
  5092.9 2213.58  5107.1 2218.44  5177.3 2232.76  5268.9 2256.57  5273.8 2256.57
#Mann= 4 ,-1 , 0
  4752.3     .07       0  4873.3     .16       0  5041.5     .07       0
  5045.5     .16       0
Bank Sta=5041.5,5045.5
XS Rating Curve= 0 ,0
Exp/Cntr=0.3,0.1

Type RM Length L Ch R = 1 ,17297   ,69,69,69
BEGIN DESCRIPTION:
Elm 74 17296.7
END DESCRIPTION:
XS GIS Cut Line= 3
      1526120.57      6760994.93      1526315.86      6760853.89
      1526471.01      6760664.26
#Sta/Elev= 30
  4755.7 2239.37  4777.9 2238.22  4825.7 2231.63  4863.7 2220.03  4878.4 2212.29
  4893.2 2208.29  4934.9 2204.94  4958.2 2204.74  4964.3 2201.57  4970.9 2195.31
    4979 2189.86  4985.2 2189.06    4991 2185.68  4991.2 2185.18    4995 2185.68
  5000.4 2185.69  5006.9 2188.94  5014.8 2186.79  5021.3 2193.28  5029.1 2189.29
  5035.6 2197.57    5050 2193.16  5056.4 2201.08  5070.8  2205.7  5085.1 2206.52
  5107.4 2212.78  5113.8 2213.01  5171.3 2224.98  5235.2 2244.04  5241.6 2247.11
#Mann= 4 ,-1 , 0
  4755.7     .07       0  4825.7     .16       0    4991     .07       0
    4995     .16       0
Bank Sta=4991,4995
XS Rating Curve= 0 ,0
Exp/Cntr=0.3,0.1

Type RM Length L Ch R = 1 ,17228   ,106,106,106
BEGIN DESCRIPTION:
Elm 74 17227.55
END DESCRIPTION:
XS GIS Cut Line= 3
      1526133.53      6761029.69      1526365.77      6760901.63
       1526524.2      6760678.09
#Sta/Elev= 30
  4733.3 2236.36  4743.9 2233.82  4749.6 2235.11  4765.7 2231.32  4771.4 2233.14
  4788.3 2226.78  4793.2 2228.24  4809.3 2223.76    4830 2221.95  4847.1 2213.69
  4860.6 2211.15  4928.5 2203.64  4940.5 2196.84  4950.3 2195.29    4956 2192.12
  4984.2 2184.07  4984.5 2183.57  4988.2 2184.07  4993.8 2190.17  4997.1 2195.58
  5002.2 2195.58  5007.5 2200.15  5022.2 2205.01  5078.8  2205.3  5114.5 2208.45
  5137.8 2213.73    5144 2217.04  5223.6 2236.73    5245 2244.31  5272.5 2250.75
#Mann= 5 ,-1 , 0
  4733.3     .07       0  4788.3    .035       0    4830     .16       0
  4984.2     .07       0  4988.2     .16       0
Bank Sta=4984.2,4988.2
XS Rating Curve= 0 ,0
Exp/Cntr=0.3,0.1

Type RM Length L Ch R = 1 ,17122   ,110,110,110
BEGIN DESCRIPTION:
Elm 74 17121.75
END DESCRIPTION:
XS GIS Cut Line= 3
      1526137.89       6761086.1      1526411.34      6760992.78
      1526586.65      6760722.25
#Sta/Elev= 30
  4709.4 2241.55  4753.6  2239.6  4783.3 2235.47  4801.4  2229.2  4809.3 2223.53
  4814.6    2224  4840.6 2206.87  4859.2 2204.72  4949.4    2202  4959.9 2198.98
  4971.2 2189.86  4989.6 2182.07  4989.9 2181.57  4993.6 2182.07  4997.3 2187.68
  5027.3 2193.38  5033.2 2191.68  5048.4 2199.33  5054.3  2196.9  5063.5 2201.05
  5069.5 2197.83  5084.7 2206.02  5090.6 2201.91  5105.8 2206.67  5111.7  2204.1
  5235.7 2223.74  5308.2 2245.14  5314.1 2242.44  5318.3 2244.59  5320.7 2245.82
#Mann= 6 ,-1 , 0
  4709.4     .07       0  4753.6    .035       0  4859.2     .16       0
  4989.6     .07       0  4993.6     .16       0  5318.3     .07       0
Bank Sta=4989.6,4993.6
XS Rating Curve= 0 ,0
Exp/Cntr=0.3,0.1

Type RM Length L Ch R = 1 ,17012   ,85,85,85
BEGIN DESCRIPTION:
Elm 74 17012.11
END DESCRIPTION:
XS GIS Cut Line= 3
      1526218.23      6761188.08       1526487.3       6761070.9
      1526760.37      6760849.85
#Sta/Elev= 30
  4705.7 2239.29    4713  2238.4  4718.5 2234.08  4734.9 2235.21  4768.8 2226.44
  4788.8 2220.34  4800.3 2213.25  4823.1 2207.85  4876.7 2202.23  4931.2 2200.55
  4958.1 2192.26  4963.7 2191.64  4974.8 2183.25  4983.8 2180.32    4984 2179.82
  4987.8 2180.32  5007.2 2186.44    5028 2197.36  5056.8 2198.53    5092 2209.07
  5106.3 2206.18  5127.1 2209.28  5135.1 2205.71  5141.5 2208.51  5149.5 2205.44
  5163.5 2206.73  5273.6 2229.31    5305 2239.85  5326.9 2251.77  5350.5 2258.02
#Mann= 6 ,-1 , 0
  4705.7     .07       0  4768.8    .035       0  4958.1     .16       0
  4983.8     .07       0  4987.8     .16       0  5273.6     .07       0
Bank Sta=4983.8,4987.8
XS Rating Curve= 0 ,0
Exp/Cntr=0.3,0.1

Type RM Length L Ch R = 1 ,16927   ,77,77,77
BEGIN DESCRIPTION:
Elm 74 16926.8
END DESCRIPTION:
XS GIS Cut Line= 3
      1526357.08      6761290.09      1526554.57      6761125.16
      1526793.31      6760843.01
#Sta/Elev= 30
    4750 2231.21  4827.7 2217.92  4849.8 2220.44  4864.1 2218.02  4870.7 2213.57
    4885 2215.58  4891.5 2211.73  4901.3 2212.79  4905.8 2209.68  4913.6 2211.66
  4920.1  2207.1  4927.9 2208.25  4934.4  2203.3  4942.2 2204.57  4948.8 2201.54
  4963.1 2205.02  4977.4 2198.87  4983.9  2191.6  5002.3 2179.21  5002.6 2178.71
  5006.3 2179.21  5038.5 2193.31  5126.1  2197.7  5154.6  2212.4  5168.9 2215.35
  5204.1 2210.59  5239.4 2224.11    5303 2241.76  5331.5 2257.08  5376.9 2262.12
#Mann= 6 ,-1 , 0
    4750     .07       0  4901.3    .035       0  5002.3    .035       0
  5006.3    .035       0  5038.5     .16       0    5303     .07       0
Bank Sta=5002.3,5006.3
XS Rating Curve= 0 ,0
Exp/Cntr=0.3,0.1

Type RM Length L Ch R = 1 ,16850   ,63,63,63
BEGIN DESCRIPTION:
Elm 74 16850.34
END DESCRIPTION:
XS GIS Cut Line= 3
      1526385.29      6761313.97      1526589.29       6761172.9
       1526834.5       6760927.7
#Sta/Elev= 30
  4703.2 2231.65  4763.7 2225.29    4808 2222.67  4850.2 2220.16  4900.9 2212.35
  4930.7 2210.38  4936.7 2205.84  4945.5 2202.15  4951.1 2193.44  4958.7 2189.12
  4965.8 2179.96  4970.9 2178.75  4971.1 2178.25  4974.9 2178.75  5001.2 2181.57
  5008.2 2184.98  5029.4 2184.88  5036.5 2187.09  5043.6 2186.09  5050.7 2190.49
  5057.7 2189.18  5064.8 2192.98  5100.2 2196.25  5107.2 2198.54  5142.6 2203.13
  5163.8 2210.17  5213.3 2232.29  5248.6 2243.86    5284 2260.91    5298 2262.39
#Mann= 5 ,-1 , 0
  4703.2     .07       0    4808    .035       0  4930.7     .16       0
  4970.9     .07       0  4974.9     .16       0
Bank Sta=4970.9,4974.9
XS Rating Curve= 0 ,0
Exp/Cntr=0.3,0.1

Type RM Length L Ch R = 1 ,16787   ,92,92,92
BEGIN DESCRIPTION:
Elm 74 16786.88
END DESCRIPTION:
XS GIS Cut Line= 3
      1526389.64      6761353.02      1526691.29      6761136.01
      1526910.04      6760912.98
#Sta/Elev= 30
  4633.4 2234.26  4732.8 2224.13  4870.5 2211.83  4912.9 2204.36  4920.9 2203.39
    4927 2197.09  4935.6 2198.33  4941.7 2184.49  4956.5 2188.58  4962.6 2178.17
  4971.2 2180.66  4975.3 2176.76  4975.6 2176.26  4979.3 2176.76  5062.8 2185.74
  5069.9 2190.29  5076.9 2188.16    5084 2196.72  5091.1 2195.35  5098.2 2201.19
  5105.2 2201.46  5112.3 2207.69  5119.3 2209.11  5126.5 2214.41  5168.9 2232.62
  5190.1 2237.99  5225.5 2255.85  5239.6 2259.89  5268.7 2261.75  5317.4 2262.87
#Mann= 6 ,-1 , 0
  4633.4     .07       0  4732.8    .035       0  4912.9     .16       0
  4975.3     .07       0  4979.3     .16       0  5268.7     .07       0
Bank Sta=4975.3,4979.3
XS Rating Curve= 0 ,0
Exp/Cntr=0.3,0.1

Type RM Length L Ch R = 1 ,16695   ,149,149,149
BEGIN DESCRIPTION:
Elm 74 16694.59
END DESCRIPTION:
XS GIS Cut Line= 3
      1526424.36      6761363.87      1526760.74      6761192.43
      1527101.78      6761140.63
#Sta/Elev= 30
  4630.9 2230.43    4681 2224.64  4762.8 2220.25  4807.3 2212.51    4874 2204.22
  4879.6  2206.8  4912.2 2198.88  4918.5 2195.71  4934.7 2194.19  4940.7 2190.99
  4946.3 2192.68  4957.1  2188.7  4962.9 2182.69  4990.8 2181.56  5005.7 2177.89
  5020.9 2174.07  5021.1 2173.57  5024.9 2174.07  5043.1 2179.97  5093.7  2189.8
  5133.5 2214.95  5138.5 2211.71  5144.2 2218.05  5194.8 2236.51  5202.2 2241.44
  5207.2 2239.08  5225.2 2250.47  5235.3 2254.01  5270.8 2263.66  5353.4 2279.19
#Mann= 5 ,-1 , 0
  4630.9     .07       0    4681    .035       0  5005.7     .16       0
  5020.9    .035       0  5024.9     .16       0
Bank Sta=5020.9,5024.9
XS Rating Curve= 0 ,0
Exp/Cntr=0.3,0.1

Type RM Length L Ch R = 1 ,16546   ,129,129,129
BEGIN DESCRIPTION:
Elm 74 16545.58
END DESCRIPTION:
XS GIS Cut Line= 3
       1526456.9      6761411.62      1526760.74      6761344.34
      1527077.56       6761209.8
#Sta/Elev= 30
  4685.8 2225.03  4696.2 2223.31  4810.4 2221.52  4827.2 2220.15  4847.7 2214.06
  4868.9 2210.45  4929.7 2204.55  4956.1 2200.58  4961.2 2197.73  4970.6 2196.39
  4991.1 2189.92  4996.6  2182.9  5002.6 2178.45  5010.5 2171.83  5010.7 2171.33
  5014.5 2171.83    5022  2172.3  5034.2 2177.24  5066.8 2182.57  5074.7 2185.05
  5088.5 2193.45  5156.5 2205.82  5180.2 2213.07  5186.3  2216.9  5227.5 2225.56
  5240.6 2232.18  5251.2 2235.79  5262.4  2244.7    5295  2260.6  5341.2 2269.08
#Mann= 6 ,-1 , 0
  4685.8     .07       0  4696.2    .063       0  4810.4    .035       0
  5002.6     .16       0  5010.5    .035       0  5014.5     .16       0
Bank Sta=5010.5,5014.5
XS Rating Curve= 0 ,0
Exp/Cntr=0.3,0.1

Type RM Length L Ch R = 1 ,16417   ,104,104,104
BEGIN DESCRIPTION:
Elm 74 16416.53
END DESCRIPTION:
XS GIS Cut Line= 3
      1526500.36      6761465.87      1526854.05      6761437.66
      1527121.56      6761355.68
#Sta/Elev= 30
  4648.9 2222.84    4784 2221.12  4812.9 2212.82  4854.2 2202.95  4894.3 2203.52
  4912.4  2200.1    4938 2188.34  4954.5 2176.14  4982.6 2170.64  4982.9 2170.14
  4986.6 2170.64  4994.6 2174.34  5001.7 2182.05  5006.8 2182.05  5014.8 2188.88
    5058 2199.11  5077.9 2201.62  5085.5 2205.56  5090.7 2204.87  5118.3 2215.79
  5123.5 2215.93  5156.2 2229.26  5161.6 2233.32  5194.2 2244.17  5215.6 2254.62
  5221.8 2258.14  5245.3 2263.89  5254.5 2265.92  5259.7 2264.39  5283.5 2273.96
#Mann= 6 ,-1 , 0
  4648.9    .063       0  4812.9    .035       0  4912.4     .16       0
  4982.6     .07       0  4986.6     .16       0  5215.6     .07       0
Bank Sta=4982.6,4986.6
XS Rating Curve= 0 ,0
Exp/Cntr=0.3,0.1

Type RM Length L Ch R = 1 ,16313   ,131,131,131
BEGIN DESCRIPTION:
Elm 74 16312.71
END DESCRIPTION:
XS GIS Cut Line= 3
      1526485.13      6761524.46      1526851.88      6761541.82
      1527086.24      6761476.72
#Sta/Elev= 30
  4630.4 2226.94  4720.4 2221.81  4800.5 2221.17    4807 2218.95  4813.2 2218.12
  4820.5 2214.07  4870.5 2198.63  4880.6 2197.07    4906 2198.11  4920.6 2197.37
  4940.6 2192.14  4980.7 2174.54  4996.6 2169.64  5009.2 2168.88  5009.4 2168.38
  5013.2 2168.88  5021.6 2173.43  5028.6 2182.48  5033.8 2185.08  5073.5 2191.94
  5107.5 2207.54  5125.3 2218.82  5141.8 2232.69    5147 2233.83    5176 2253.04
  5181.2 2252.44  5187.6 2256.98  5215.5 2264.89  5220.6 2264.22  5240.8 2268.68
#Mann= 5 ,-1 , 0
  4630.4    .063       0    4807    .035       0    4906     .16       0
  5009.2     .07       0  5013.2     .16       0
Bank Sta=5009.2,5013.2
XS Rating Curve= 0 ,0
Exp/Cntr=0.3,0.1

Type RM Length L Ch R = 1 ,16182   ,104,104,104
BEGIN DESCRIPTION:
Elm 74 16182.49
END DESCRIPTION:
XS GIS Cut Line= 3
      1526478.64      6761624.29      1526851.88      6761672.03
      1527091.42      6761615.93
#Sta/Elev= 30
  4620.9 2223.79  4702.6    2221  4748.3 2219.37  4845.6 2203.98  4879.3 2200.66
  4899.5  2199.7  4925.3 2201.17  4939.8 2198.95  4949.9 2194.24  4980.2 2172.73
  4990.2 2171.08  4994.2 2166.95  4994.5 2166.45  4998.2 2166.95  5001.4 2166.95
  5010.7    2170  5020.9 2180.58  5031.2 2184.29  5072.3 2184.87  5092.8  2186.9
  5113.4 2190.79  5126.6  2196.6  5144.2 2207.23    5164 2223.04  5169.1 2225.44
    5175 2232.09  5205.8 2249.69  5211.6 2255.85  5226.3 2261.53  5243.2 2265.26
#Mann= 4 ,-1 , 0
  4620.9    .063       0  4702.6     .16       0  4994.2     .07       0
  4998.2     .16       0
Bank Sta=4994.2,4998.2
XS Rating Curve= 0 ,0
Exp/Cntr=0.3,0.1

Type RM Length L Ch R = 1 ,16078   ,132,132,132
BEGIN DESCRIPTION:
Elm 74 16077.82
END DESCRIPTION:
XS GIS Cut Line= 3
      1526428.72      6761752.33      1526854.05       6761776.2
      1527111.13      6761737.31
#Sta/Elev= 30
  4573.1 2221.82  4579.4 2218.99  4601.8 2216.35  4639.5 2211.22  4669.5 2202.74
  4700.8 2207.48  4709.6 2208.84  4729.6 2207.73  4769.7 2201.78  4869.8 2197.89
  4899.9    2200  4943.5 2197.55    4960 2194.08    4980 2182.16  4997.1 2167.93
  5002.1 2167.93  5008.2  2164.6  5008.4  2164.1  5012.2  2164.6  5040.5 2178.76
  5050.6  2182.3  5101.2 2183.68  5121.4 2188.63  5141.6 2197.13  5150.5 2205.62
  5155.5 2204.88  5182.1 2222.24  5219.3 2242.01  5252.9 2251.81  5259.1 2254.94
#Mann= 5 ,-1 , 0
  4573.1     .07       0  4601.8    .063       0  4700.8     .16       0
  5008.2     .07       0  5012.2     .16       0
Bank Sta=5008.2,5012.2
XS Rating Curve= 0 ,0
Exp/Cntr=0.3,0.1

Type RM Length L Ch R = 1 ,15946   ,109,109,109
BEGIN DESCRIPTION:
Elm 74 15945.68
END DESCRIPTION:
XS GIS Cut Line= 3
        1526496.      6761854.33      1526901.79      6761893.39
      1527144.81      6761841.31
#Sta/Elev= 30
  4593.2 2227.51  4602.2 2225.66  4622.3 2225.52  4650.8 2221.33  4681.5 2215.14
  4685.7 2216.77  4712.8 2203.27  4732.8 2196.58  4943.8 2182.54  4953.9  2180.7
    4984 2163.57  4992.9 2164.12    4996 2162.78  4996.2 2162.28    5000 2162.78
    5006 2167.89  5014.4 2168.59  5050.3 2180.91  5094.6 2189.85  5137.1 2212.55
  5144.1 2218.09  5149.2 2215.78  5150.5 2216.47  5167.8 2225.52  5188.2 2232.51
  5193.5 2235.94  5237.8 2241.74  5242.9 2244.25    5247 2249.15  5249.4 2249.15
#Mann= 6 ,-1 , 0
  4593.2     .07       0  4650.8    .063       0  4681.5     .16       0
    4996     .07       0    5000     .16       0  5150.5     .07       0
Bank Sta=4996,5000
XS Rating Curve= 0 ,0
Exp/Cntr=0.3,0.1

Type RM Length L Ch R = 1 ,15837   ,141,141,141
BEGIN DESCRIPTION:
Elm 74 15837.29
END DESCRIPTION:
XS GIS Cut Line= 3
      1526478.65      6761967.17      1526914.82      6762001.89
      1527157.83      6761934.63
#Sta/Elev= 30
  4572.8 2229.33  4639.4 2225.41  4719.6 2217.25  4739.7 2211.04  4759.7 2201.56
  4799.9 2191.91    4830 2186.38  4970.4 2177.81  4990.5 2167.66  5005.9 2161.48
  5006.2 2160.98  5009.9 2161.48    5013 2161.48  5020.9 2165.36  5040.1 2176.97
  5045.3 2177.35    5052 2180.51  5072.8 2183.36  5119.1 2193.13  5124.7 2197.54
  5145.6 2207.51  5153.4 2212.15  5166.2 2216.67  5192.9 2220.11  5198.1 2222.95
  5227.2 2223.89  5232.4 2226.33  5238.8 2225.74  5258.5 2231.16  5262.5 2231.16
#Mann= 4 ,-1 , 0
  4572.8     .16       0  5005.9     .07       0  5009.9     .16       0
  5145.6     .07       0
Bank Sta=5005.9,5009.9
XS Rating Curve= 0 ,0
Exp/Cntr=0.3,0.1

Type RM Length L Ch R = 1 ,15696   ,149,149,149
BEGIN DESCRIPTION:
Elm 74 15695.64
END DESCRIPTION:
XS GIS Cut Line= 3
      1526604.53      6762099.56      1526906.13      6762142.95
      1527121.61      6762069.69
#Sta/Elev= 30
  4696.9 2214.98  4716.8 2211.39  4737.8 2205.43  4787.3 2196.24  4798.4 2192.67
  4828.7 2194.71  4857.7 2189.84  4862.8 2190.41  4879.2 2185.42  4909.5 2169.64
  4928.2 2165.94  4960.1 2165.46  4988.4 2160.07  4988.6 2159.57  4992.4 2160.07
  5003.7 2161.69  5029.7 2173.69  5066.3 2177.06  5084.9 2180.93  5097.7 2186.62
    5106 2191.95  5123.8 2197.64  5129.1 2202.23  5137.7 2203.37  5155.2 2201.04
  5160.5 2205.91    5180 2204.44  5186.6 2207.43  5201.1 2207.51  5229.2 2213.15
#Mann= 3 ,-1 , 0
  4696.9     .16       0  4988.4     .07       0  4992.4     .16       0
Bank Sta=4988.4,4992.4
XS Rating Curve= 0 ,0
Exp/Cntr=0.3,0.1

Type RM Length L Ch R = 1 ,15547   ,121,121,121
BEGIN DESCRIPTION:
Elm 74 15547.08
END DESCRIPTION:
XS GIS Cut Line= 3
      1526658.72      6762310.06      1526906.13      6762292.69
      1527090.29      6762199.53
#Sta/Elev= 30
  4747.1 2218.17  4753.4 2214.79  4793.5 2203.17  4823.6 2197.36  4843.8 2195.65
  4873.7 2193.06  4883.7 2191.56  4903.8 2186.73  4923.8  2184.1  4933.8 2181.81
  4943.9 2180.34  4953.9 2180.18  4963.9  2175.9    4984 2170.14  4992.9 2163.01
  4997.3 2163.01  5011.6 2157.02  5011.9 2156.52  5015.6 2157.02  5035.9 2163.25
  5049.9  2170.1  5063.8  2173.5  5102.8 2173.77    5125 2174.59  5139.5 2176.24
  5152.9 2181.28  5175.2 2191.43  5191.9 2201.05  5197.5 2202.83  5201.5 2206.05
#Mann= 4 ,-1 , 0
  4747.1     .07       0  4843.8     .16       0  5011.6     .07       0
  5015.6     .16       0
Bank Sta=5011.6,5015.6
XS Rating Curve= 0 ,0
Exp/Cntr=0.3,0.1

Type RM Length L Ch R = 1 ,15426   ,98,98,98
BEGIN DESCRIPTION:
Elm 74 15426.2
END DESCRIPTION:
XS GIS Cut Line= 3
      1526778.13      6762448.93      1526995.11      6762377.33
      1527116.64      6762253.63
#Sta/Elev= 30
  4772.6 2202.03  4788.3 2196.53  4800.9 2193.56  4844.9 2187.82  4864.1 2184.75
  4906.2  2180.9  4947.1  2174.9  4952.3 2172.45  4958.9 2164.85  4969.4 2156.36
  4976.8 2156.16  4977.1 2155.66  4980.8 2156.16  4984.1 2157.73  5004.1  2159.6
  5014.6 2161.91  5021.8 2163.79  5028.8 2168.03  5042.9 2171.89  5092.5 2174.66
  5099.5 2176.53  5106.6 2176.58  5113.6 2180.35  5120.8  2180.9  5127.8 2185.04
  5134.9 2185.91  5141.9 2190.49    5149 2192.25  5169.8 2202.03  5174.5 2202.03
#Mann= 4 ,-1 , 0
  4772.6     .07       0  4844.9     .16       0  4976.8     .07       0
  4980.8     .16       0
Bank Sta=4976.8,4980.8
XS Rating Curve= 0 ,0
Exp/Cntr=0.3,0.1

Type RM Length L Ch R = 1 ,15328   ,186,186,186
BEGIN DESCRIPTION:
Elm 74 15327.93
END DESCRIPTION:
XS GIS Cut Line= 3
      1526823.65      6762563.97      1527073.24      6762442.43
      1527175.21      6762327.44
#Sta/Elev= 30
  4733.1 2202.25  4737.7 2203.67  4827.9 2194.45  4844.9 2187.87  4850.5  2188.9
  4852.4 2187.83  4867.4 2181.08    4873 2181.42  4879.2 2177.21  4923.7  2172.7
  4957.1 2162.18  4991.3 2155.11  4999.5 2154.86  4999.8 2154.36  5003.5 2154.86
  5010.7 2161.39  5015.8 2161.39  5036.3 2171.89  5057.2 2176.09  5064.8 2175.82
  5071.4  2177.8  5107.4 2181.78  5114.1 2184.33  5121.6 2184.74  5128.3 2188.34
  5135.9 2188.75  5142.5 2192.98  5150.1 2192.25  5156.8 2197.08  5164.4 2197.19
#Mann= 4 ,-1 , 0
  4733.1     .07       0  4852.4     .16       0  4999.5     .07       0
  5003.5     .16       0
Bank Sta=4999.5,5003.5
XS Rating Curve= 0 ,0
Exp/Cntr=0.3,0.1

Type RM Length L Ch R = 1 ,15142   ,78,78,78
BEGIN DESCRIPTION:
Elm 74 15141.57
END DESCRIPTION:
XS GIS Cut Line= 3
      1526875.78      6762744.07      1527164.38      6762596.51
      1527324.86       6762472.9
#Sta/Elev= 30
    4675 2216.13  4695.1 2213.32  4707.8  2213.4  4717.4  2210.6    4723 2210.95
  4730.3  2208.3  4745.2 2205.83  4767.4 2200.12    4784 2194.16  4797.7 2190.51
  4842.6 2180.85  4850.6 2180.54  4905.5 2172.97  4939.5 2168.81  4967.3 2167.42
  4977.4 2162.52  4983.9 2154.35  4987.5 2151.51  4987.8 2151.01  4991.5 2151.51
    5002 2152.48  5034.6 2157.65  5040.9 2160.31  5055.4 2163.73  5084.4 2176.66
  5098.9 2181.17    5155 2187.02    5184 2188.59  5198.6 2190.71  5201.7 2191.87
#Mann= 4 ,-1 , 0
    4675     .07       0  4905.5     .16       0  4987.5     .07       0
  4991.5     .16       0
Bank Sta=4987.5,4991.5
XS Rating Curve= 0 ,0
Exp/Cntr=0.3,0.1

Type RM Length L Ch R = 1 ,15064   ,74,74,74
BEGIN DESCRIPTION:
Elm 74 15063.5
END DESCRIPTION:
XS GIS Cut Line= 3
       1526919.2      6762759.26      1527218.63      6762652.94
      1527327.17      6762533.55
#Sta/Elev= 30
  4680.4 2207.49  4686.6 2205.17  4700.8 2205.32  4739.6 2196.14  4762.5 2192.78
  4788.1 2186.67  4813.6 2184.48  4893.2 2170.78  4930.6 2165.48  4962.5 2162.56
  4967.9 2160.11  4973.2 2156.11  4993.5 2153.53  5003.9 2150.66  5004.1 2150.16
  5007.9 2150.66  5013.3    2151  5020.1 2156.62  5027.5 2160.02  5034.3 2165.35
  5041.7 2168.35  5048.5 2173.93  5055.9 2175.66  5062.6    2180  5098.5 2181.22
  5121.7 2177.75  5133.6  2180.2  5140.4 2180.09  5154.2 2183.28  5159.5 2183.28
#Mann= 5 ,-1 , 0
  4680.4     .07       0  4893.2     .16       0  5003.9     .07       0
  5007.9     .16       0  5121.7     .07       0
Bank Sta=5003.9,5007.9
XS Rating Curve= 0 ,0
Exp/Cntr=0.3,0.1

Type RM Length L Ch R = 1 ,14990   ,138,138,138
BEGIN DESCRIPTION:
Elm 74 14990.08
END DESCRIPTION:
XS GIS Cut Line= 3
      1526947.37      6762850.42      1527270.72      6762705.02
      1527368.38      6762544.42
#Sta/Elev= 30
  4644.1 2195.04  4660.1 2190.52  4665.6 2191.93  4683.2 2189.32  4688.7 2190.29
  4758.2 2180.35  4786.8 2178.85  4804.5 2175.02    4810 2176.53  4833.1 2175.12
  4879.4 2167.81  4902.6 2167.72  4915.6  2164.8  4970.4 2161.44  4977.5 2157.59
  4998.2 2151.49  5012.6 2149.97  5012.9 2149.47  5016.6 2149.97    5042 2164.01
  5072.7 2176.88  5088.2 2175.84  5094.1 2173.13  5109.5 2173.79  5115.4 2171.69
  5146.3 2174.15  5152.2 2171.34  5167.7 2172.73  5173.5 2171.02  5186.6 2171.26
#Mann= 3 ,-1 , 0
  4644.1     .07       0  5012.6     .07       0  5016.6     .07       0
Bank Sta=5012.6,5016.6
XS Rating Curve= 0 ,0
Exp/Cntr=0.3,0.1

Type RM Length L Ch R = 1 ,14852   ,76,76,76
BEGIN DESCRIPTION:
Elm 74 14851.93
END DESCRIPTION:
XS GIS Cut Line= 3
      1527147.02      6762948.07      1527359.69      6762807.02
      1527555.03       6762624.7
#Sta/Elev= 30
  4750.5  2181.1  4756.9 2181.24  4762.9 2177.74    4799 2173.49    4808 2173.39
  4856.1 2165.84  4907.2 2162.51  4937.3 2159.25  4979.4 2157.62  4988.1 2155.26
  4994.5 2150.52  5000.3 2148.21  5005.7 2148.21  5006.9 2146.85  5007.1 2146.35
  5010.9 2146.85  5029.9  2153.1  5037.2 2157.79    5044 2159.05  5079.7 2163.46
    5129 2173.79  5143.2 2174.88    5150 2177.22  5178.4 2178.98  5185.7  2178.2
  5192.5 2179.82  5199.9  2178.7    5214 2180.16  5256.5 2190.51  5272.9 2192.93
#Mann= 3 ,-1 , 0
  4750.5     .07       0  5006.9     .07       0  5010.9     .07       0
Bank Sta=5006.9,5010.9
XS Rating Curve= 0 ,0
Exp/Cntr=0.3,0.1

Type RM Length L Ch R = 1 ,14776   ,217,217,217
BEGIN DESCRIPTION:
Elm 74 14776.35
END DESCRIPTION:
XS GIS Cut Line= 3
      1527162.21      6762989.31      1527387.91      6762876.46
      1527633.14      6762635.57
#Sta/Elev= 30
  4744.1 2190.43  4755.5 2190.43  4769.6 2186.34  4777.9 2187.52  4783.5 2184.41
  4800.2 2189.61  4805.8 2186.35  4814.3 2186.66  4822.6 2185.13  4828.2 2180.39
    4845 2175.72  4850.5 2171.78  4867.3 2170.04  4872.9 2166.83  4889.7 2165.54
  4895.3 2162.91  4926.1 2158.58  4962.3 2155.65  4979.1 2149.94  5005.4 2145.35
  5005.6 2144.85  5009.4 2145.35  5042.8 2157.81    5064 2160.57  5071.1 2163.24
  5099.4 2166.95  5148.8 2170.64  5290.3 2184.67  5332.7 2192.99  5340.2 2193.32
#Mann= 3 ,-1 , 0
  4744.1     .07       0  5005.4     .07       0  5009.4     .07       0
Bank Sta=5005.4,5009.4
XS Rating Curve= 0 ,0
Exp/Cntr=0.3,0.1

Type RM Length L Ch R = 1 ,14559   ,127,127,127
BEGIN DESCRIPTION:
Elm 74 14559.24
END DESCRIPTION:
XS GIS Cut Line= 3
      1527357.54      6763095.64      1527552.84      6763024.03
      1527785.04      6762820.03
#Sta/Elev= 30
  4801.1 2189.66  4830.3 2183.56  4842.1 2179.04  4867.2  2174.1    4873 2171.57
  4892.4 2170.37  4897.7 2167.27  4908.3 2166.47  4915.6 2165.66  4931.5 2160.41
  4947.5  2158.7  4968.8 2153.27  4978.6 2153.01  4990.1  2149.9  5000.8 2149.25
  5007.6 2146.83  5014.7 2142.07  5020.2 2141.74  5020.5 2141.24  5024.2 2141.74
  5043.1 2151.99  5053.2 2155.68  5106.7 2158.61  5120.9 2160.47  5128.5    2160
    5157 2162.94  5198.7 2169.76    5249 2179.89  5298.4 2185.59  5318.2 2186.45
#Mann= 5 ,-1 , 0
  4801.1     .07       0  4908.3     .16       0  5020.2     .07       0
  5024.2     .16       0  5053.2     .07       0
Bank Sta=5020.2,5024.2
XS Rating Curve= 0 ,0
Exp/Cntr=0.3,0.1

Type RM Length L Ch R = 1 ,14432   ,194,194,194
BEGIN DESCRIPTION:
Elm 74 14432.31
END DESCRIPTION:
XS GIS Cut Line= 3
      1527407.41      6763147.73      1527633.13      6763117.35
      1527865.36      6762987.12
#Sta/Elev= 30
    4771 2180.37  4806.6 2175.13  4829.1 2170.56  4869.5 2170.37  4955.8 2162.67
  4970.4 2159.97  4990.5 2151.45  4997.2 2144.22  5002.7 2144.22  5005.1 2140.28
  5005.4 2139.78  5009.1 2140.28  5012.9 2140.45  5028.8 2146.25  5044.8 2148.18
  5050.5 2151.57  5072.2 2153.65  5104.1 2154.36  5121.6 2159.78  5147.5 2169.86
  5153.2  2173.2  5169.2 2177.93  5174.9 2182.18  5190.9 2185.45  5196.6  2188.8
  5218.7 2191.18  5228.5 2188.73  5234.2 2191.44  5241.7 2193.02    5265 2194.61
#Mann= 5 ,-1 , 0
    4771     .07       0  4806.6     .16       0  5005.1     .07       0
  5009.1     .16       0  5121.6     .07       0
Bank Sta=5005.1,5009.1
XS Rating Curve= 0 ,0
Exp/Cntr=0.3,0.1

Type RM Length L Ch R = 1 ,14238   ,99,99,99
BEGIN DESCRIPTION:
Elm 74 14237.93
END DESCRIPTION:
XS GIS Cut Line= 3
      1527463.84      6763173.77      1527739.47      6763219.34
      1527965.13      6763115.19
#Sta/Elev= 30
  4652.9 2173.61  4785.8 2169.47  4826.4 2166.38  4836.8 2163.94  4856.8 2162.93
  4866.9 2161.12  4887.2 2155.68  4892.8 2152.59  4897.9  2153.9  4907.5 2152.28
  4945.6 2149.93  4968.6 2142.37  4974.1 2139.22  4989.5 2138.89  4989.8 2138.39
  4993.5 2138.89    4997 2141.98    5020 2145.77  5037.4 2152.49  5059.5 2158.21
  5065.9  2162.2  5081.5 2167.35  5088.8 2171.56  5094.3 2172.57  5111.8 2180.85
  5117.3 2181.61  5134.7 2189.94  5139.1 2190.52  5147.6 2192.69  5180.8 2192.56
#Mann= 4 ,-1 , 0
  4652.9     .16       0  4989.5     .07       0  4993.5     .16       0
  5139.1     .07       0
Bank Sta=4989.5,4993.5
XS Rating Curve= 0 ,0
Exp/Cntr=0.3,0.1

Type RM Length L Ch R = 1 ,14139   ,182,182,182
BEGIN DESCRIPTION:
Elm 74 14139.42
END DESCRIPTION:
XS GIS Cut Line= 3
      1527522.41      6763188.95      1527858.83      6763267.09
      1528054.16      6763234.53
#Sta/Elev= 30
  4657.1 2172.18  4752.2 2168.05    4783 2161.93    4803 2161.28  4808.1 2158.65
  4813.8 2158.91    4824 2157.73  4850.8 2151.77  4916.4 2149.83    4936 2144.52
  4967.7 2144.44  4983.8 2140.21  4988.9 2141.08  4997.9 2139.31  5002.5 2139.31
  5006.7    2138    5007  2137.5  5010.7    2138  5018.9    2140  5025.6  2147.3
  5030.7  2154.9  5039.1 2162.89  5049.3 2168.79  5079.7  2181.8  5086.5 2185.94
  5091.5 2185.24  5110.1 2189.27  5152.4 2191.32  5170.9 2191.59  5200.5 2188.74
#Mann= 3 ,-1 , 0
  4657.1     .16       0  5006.7     .07       0  5010.7     .16       0
Bank Sta=5006.7,5010.7
XS Rating Curve= 0 ,0
Exp/Cntr=0.3,0.1

Type RM Length L Ch R = 1 ,13957   ,165,165,165
BEGIN DESCRIPTION:
Elm 74 13956.59
END DESCRIPTION:
XS GIS Cut Line= 3
      1527620.15      6763466.73      1527900.06      6763434.19
       1528104.1      6763390.77
#Sta/Elev= 30
  4716.3 2161.38  4721.2 2161.38  4747.5 2157.82  4752.5 2158.74  4781.6  2156.2
    4831 2148.49  4836.1 2148.93    4842 2147.93  4872.2 2147.24  4912.5 2143.19
  4962.8 2141.42    4996  2134.4  4996.3  2133.9  5000.1  2134.4    5006 2134.72
  5023.6 2151.66  5033.8 2159.44    5044 2166.05  5055.6 2172.49  5064.5 2172.14
    5095 2167.15  5100.1 2169.31  5105.4 2169.41  5125.8 2177.13  5136.1 2179.11
  5149.7 2180.95  5166.7 2180.45  5194.1 2181.64  5199.3 2183.27  5206.7    2183
#Mann= 3 ,-1 , 0
  4716.3     .16       0    4996     .07       0  5000.1     .16       0
Bank Sta=4996,5000.1
XS Rating Curve= 0 ,0
Exp/Cntr=0.3,0.1
