HEC-RAS study Elm 76.prj: Elm 76 Base Level Engineering

--- Elm 76.g01 (geometry) --- (continued)

Type RM Length L Ch R = 1,4898,89,89,89
BEGIN DESCRIPTION:
Elm 76 4898.16
END DESCRIPTION:
XS GIS Cut Line= 3
      1529859.29      6761568.28      1530071.50      6761445.90
      1530307.19      6761303.97
#Sta/Elev= 30
  4762.2 2187.20  4767.6 2187.37  4789.5 2186.96  4819.7 2178.63  4893.9 2161.65
  4956.1 2150.65  5010.0 2147.27  5028.5 2141.44  5028.7 2140.94  5032.5 2141.44
  5057.9 2158.27  5067.4 2161.41  5088.7 2162.41  5094.6 2165.14  5104.3 2160.35
  5110.5 2163.59  5125.6 2154.09  5131.5 2157.44  5139.7 2151.39  5152.8 2149.51
  5162.5 2154.68  5168.4 2150.69  5174.7 2157.93  5183.9 2160.93  5189.7 2158.53
  5205.3 2163.51  5248.0 2167.72  5263.5 2173.91  5269.3 2172.24  5282.3 2175.68
#Mann=7,-1,0
  4762.2    0.07       0  4767.6    0.16       0  4819.7    0.07       0
  4893.9    0.16       0  5028.5    0.07       0  5032.5    0.16       0
  5110.5    0.07       0
Bank Sta=5028.5,5032.5
Exp/Cntr=0.3,0.1

Type RM Length L Ch R = 1,4809,96,96,96
BEGIN DESCRIPTION:
Elm 76 4808.84
END DESCRIPTION:
XS GIS Cut Line= 3
      1529895.69      6761603.47      1530105.35      6761524.03
      1530296.75      6761393.82
#Sta/Elev= 30
  4776.5 2187.01  4779.5 2185.50  4786.5 2186.81  4818.5 2184.53  4834.4 2176.56
  4839.9 2169.85  4850.6 2170.16  4859.2 2174.47  4864.6 2172.19  4882.7 2175.72
  4904.1 2165.12  4925.5 2156.95  4938.5 2153.99  4968.3 2147.27  4974.5 2141.98
  4977.8 2141.07  4978.1 2140.57  4981.8 2141.07  4997.8 2146.71  5004.4 2147.23
  5019.4 2154.82  5061.3 2157.60  5076.3 2155.50  5091.2 2147.01  5097.3 2146.28
  5112.2 2152.44  5121.1 2152.30  5153.2 2159.10  5184.0 2163.87  5232.2 2167.68
#Mann=5,-1,0
  4776.5    0.07       0  4938.5    0.16       0  4977.8    0.07       0
  4981.8    0.16       0  5153.2    0.07       0
Bank Sta=4977.8,4981.8
Exp/Cntr=0.3,0.1

Type RM Length L Ch R = 1,4713,105,105,105
BEGIN DESCRIPTION:
Elm 76 4713.11
END DESCRIPTION:
XS GIS Cut Line= 3
      1529984.26      6761693.30      1530131.40      6761611.27
      1530279.85      6761479.74
#Sta/Elev= 30
  4834.3 2186.67  4919.0 2184.85  4940.8 2179.60  4949.6 2174.97  4972.5 2155.21
  4978.5 2143.30  4984.2 2140.52  4992.5 2139.45  4992.7 2138.95  4996.5 2139.45
  5000.2 2143.65  5002.8 2144.82  5016.8 2146.21  5043.2 2145.85  5057.4 2148.24
  5064.1 2150.26  5071.6 2149.76  5078.3 2151.20  5085.8 2149.01  5092.5 2152.26
  5100.1 2148.73  5106.7 2149.56  5121.0 2148.43  5127.8 2145.94  5135.2 2144.85
  5156.1 2157.07  5163.6 2160.17  5170.3 2161.80  5177.8 2162.11  5201.1 2165.53
#Mann=4,-1,0
  4834.3    0.07       0  4992.5    0.07       0  4996.5    0.07       0
  5016.8    0.16       0
Bank Sta=4992.5,4996.5
Exp/Cntr=0.3,0.1

Type RM Length L Ch R = 1,4608,107,107,107
BEGIN DESCRIPTION:
Elm 76 4608.18
END DESCRIPTION:
XS GIS Cut Line= 3
      1530126.22      6761759.68      1530213.43      6761673.77
      1530290.14      6761508.64
#Sta/Elev= 30
  4886.4 2184.57  4929.1 2182.48  4936.2 2181.29  4943.3 2181.95  4950.4 2180.64
  4957.4 2181.54  4964.5 2178.52  4971.6 2164.64  4978.7 2157.26  4985.7 2136.94
  4999.8 2137.04  5008.8 2138.85  5015.2 2136.27  5022.6 2136.90  5026.1 2136.23
  5026.3 2135.73  5030.1 2136.23  5031.0 2136.40  5045.5 2139.67  5051.0 2136.45
  5068.3 2139.96  5081.3 2141.44  5091.2 2145.31  5136.5 2144.79  5142.5 2147.24
  5148.1 2147.49  5158.5 2153.81  5165.4 2159.32  5180.6 2163.22  5190.9 2164.27
#Mann=4,-1,0
  4886.4    0.07       0  5026.1    0.07       0  5030.1    0.07       0
  5031.0    0.16       0
Bank Sta=5026.1,5030.1
Exp/Cntr=0.3,0.1

Type RM Length L Ch R = 1,4501,88,88,88
BEGIN DESCRIPTION:
Elm 76 4500.89
END DESCRIPTION:
XS GIS Cut Line= 3
      1530179.58      6761753.19      1530299.36      6761641.22
      1530417.85      6761553.98
#Sta/Elev= 30
  4834.6 2182.77  4863.4 2180.32  4870.2 2175.17  4877.5 2172.77  4884.4 2167.28
  4891.7 2165.29  4898.5 2159.68  4905.9 2158.30  4912.7 2151.39  4920.0 2151.24
  4929.0 2147.61  4948.4 2145.75  4962.5 2142.89  4969.4 2138.81  4976.7 2138.40
  4983.5 2135.40  4988.9 2135.21  4989.1 2134.71  4992.9 2135.21  4997.3 2138.05
  5005.6 2138.78  5012.1 2142.09  5018.3 2143.41  5026.7 2149.85  5032.9 2148.80
  5041.4 2153.09  5047.6 2154.66  5127.0 2161.36  5142.6 2166.81  5145.7 2166.81
#Mann=5,-1,0
  4834.6    0.07       0  4929.0    0.16       0  4988.9    0.07       0
  4992.9    0.16       0  5142.6    0.07       0
Bank Sta=4988.9,4992.9
Exp/Cntr=0.3,0.1

Type RM Length L Ch R = 1,4413,65,65,65
BEGIN DESCRIPTION:
Elm 76 4413.21
END DESCRIPTION:
XS GIS Cut Line= 3
      1530182.18      6761783.14      1530356.66      6761703.72
      1530489.45      6761604.77
#Sta/Elev= 30
  4810.8 2179.05  4815.3 2180.56  4832.8 2178.58  4838.3 2181.11  4855.9 2178.32
  4861.4 2179.47  4878.9 2171.98  4884.4 2173.78  4901.8 2165.22  4907.5 2160.47
  4913.0 2159.91  4922.6 2155.19  4930.5 2148.76  4945.7 2141.60  4959.1 2140.11
  4967.7 2135.77  4987.7 2134.20  4987.9 2133.70  4991.7 2134.20  5005.2 2138.89
  5019.8 2148.12  5034.4 2151.65  5105.3 2157.83  5119.9 2156.43  5126.1 2159.55
  5134.5 2158.18  5139.2 2160.04  5149.1 2158.85  5155.3 2161.93  5168.1 2162.00
#Mann=5,-1,0
  4810.8    0.07       0  4922.6    0.16       0  4987.7    0.07       0
  4991.7    0.16       0  5139.2    0.07       0
Bank Sta=4987.7,4991.7
Exp/Cntr=0.3,0.1

Type RM Length L Ch R = 1,4348,128,128,128
BEGIN DESCRIPTION:
Elm 76 4347.723
END DESCRIPTION:
XS GIS Cut Line= 3
      1530204.96      6761838.02      1530354.49      6761770.18
      1530504.99      6761738.00
#Sta/Elev= 30
  4835.8 2182.25  4850.1 2180.78  4873.2 2168.98  4879.8 2164.47  4890.8 2159.73
  4896.3 2155.86  4901.8 2155.80  4919.4 2149.48  4924.9 2148.60  4942.5 2142.00
  4948.0 2142.81  4962.2 2140.31  4971.0 2139.96  4978.6 2138.17  4992.1 2132.80
  4992.4 2132.30  4996.1 2132.80  5021.0 2134.72  5030.2 2137.03  5035.3 2140.24
  5041.4 2142.21  5051.7 2143.20  5079.7 2150.54  5084.8 2147.47  5102.8 2155.00
  5123.2 2159.78  5129.2 2162.66  5134.3 2162.20  5151.4 2169.09  5153.9 2169.09
#Mann=4,-1,0
  4835.8    0.07       0  4962.2    0.16       0  4992.1    0.07       0
  4996.1    0.16       0
Bank Sta=4992.1,4996.1
Exp/Cntr=0.3,0.1

Type RM Length L Ch R = 1,4220,67,67,67
BEGIN DESCRIPTION:
Elm 76 4220
END DESCRIPTION:
XS GIS Cut Line= 3
      1530165.21      6761879.50      1530314.99      6761884.71
      1530481.51      6761829.20
#Sta/Elev= 30
  4851.1 2183.10  4880.9 2181.98  4920.9 2173.31  4930.9 2168.72  4940.9 2161.85
  4948.9 2154.35  4953.9 2153.51  4961.0 2145.94  4971.0 2139.34  4981.0 2131.20
  4989.0 2130.54  4989.2 2130.04  4993.0 2130.54  4998.5 2132.43  5003.6 2132.43
  5006.3 2137.20  5011.6 2134.20  5037.9 2138.87  5043.2 2135.70  5066.9 2140.31
  5069.6 2141.11  5074.8 2135.89  5101.2 2141.90  5106.5 2139.87  5116.9 2143.05
  5127.5 2149.11  5132.8 2153.18  5138.1 2154.11  5148.6 2158.69  5176.5 2163.41
#Mann=4,-1,0
  4851.1    0.07       0  4989.0    0.07       0  4993.0    0.07       0
  5066.9    0.16       0
Bank Sta=4989,4993
Exp/Cntr=0.3,0.1

Type RM Length L Ch R = 1,4153,83,83,83
BEGIN DESCRIPTION:
Elm 76 4153.15
END DESCRIPTION:
XS GIS Cut Line= 3
      1530186.10      6762009.70      1530357.96      6761931.58
      1530481.44      6761847.97
#Sta/Elev= 30
  4815.3 2177.16  4825.1 2173.80  4831.0 2169.12  4847.0 2163.21  4854.1 2159.18
  4869.0 2157.41  4877.2 2159.19  4882.7 2152.07  4900.2 2157.34  4905.7 2152.61
  4923.3 2151.45  4928.8 2145.80  4934.9 2143.01  4951.9 2141.14  4957.3 2133.45
  4978.4 2128.62  4978.7 2128.12  4982.4 2128.62  4989.8 2128.78  4998.0 2131.45
  5002.4 2137.86  5055.0 2136.58  5073.5 2138.33  5084.9 2139.72  5090.9 2142.95
  5105.9 2144.74  5111.9 2148.35  5120.8 2150.12  5126.9 2153.40  5153.2 2161.94
#Mann=4,-1,0
  4815.3    0.07       0  4978.4    0.07       0  4982.4    0.07       0
  5073.5    0.16       0
Bank Sta=4978.4,4982.4
Exp/Cntr=0.3,0.1

Type RM Length L Ch R = 1,4070,71,71,71
BEGIN DESCRIPTION:
Elm 76 4069.99
END DESCRIPTION:
XS GIS Cut Line= 3
      1530361.87      6762077.41      1530438.69      6761934.19
      1530503.79      6761836.52
#Sta/Elev= 30
  4841.7 2174.89  4858.5 2177.26  4864.2 2176.75  4874.7 2177.23  4886.4 2175.66
  4896.7 2173.04  4924.3 2160.98  4940.5 2151.97  4946.2 2149.51  4954.5 2143.24
  4962.4 2135.56  4968.1 2135.68  4977.2 2128.92  4984.4 2127.78  4997.2 2127.78
  4997.5 2127.28  5001.2 2127.78  5004.2 2131.59  5012.1 2132.20  5021.1 2135.95
  5026.8 2135.58  5035.7 2136.60  5048.2 2142.39  5063.2 2145.88  5071.8 2150.10
  5078.2 2154.26  5084.2 2156.03  5093.3 2160.34  5114.3 2165.22  5121.6 2165.32
#Mann=4,-1,0
  4841.7    0.07       0  4997.2    0.07       0  5001.2    0.07       0
  5026.8    0.16       0
Bank Sta=4997.2,5001.2
Exp/Cntr=0.3,0.1

Type RM Length L Ch R = 1,3999,35,35,35
BEGIN DESCRIPTION:
Elm 76 3999.15
END DESCRIPTION:
XS GIS Cut Line= 3
      1530425.66      6762064.40      1530509.00      6761935.49
      1530541.25      6761821.98
#Sta/Elev= 30
  4849.2 2165.89  4854.0 2168.16  4860.0 2163.76  4875.1 2166.29  4881.1 2160.99
  4890.3 2161.33  4896.3 2156.60  4904.4 2156.03  4926.6 2141.01  4940.2 2139.69
  4947.7 2135.20  4953.7 2138.52  4962.9 2133.20  4975.9 2128.99  4988.7 2127.51
  4996.2 2125.49  4996.5 2124.99  5000.2 2125.49  5002.7 2125.49  5005.8 2132.74
  5031.3 2136.44  5039.7 2140.22  5044.9 2139.45  5052.1 2144.92  5062.5 2149.59
  5078.8 2155.64  5084.0 2152.60  5112.7 2164.42  5117.9 2164.93  5120.7 2168.86
#Mann=4,-1,0
  4849.2    0.07       0  4988.7    0.16       0  4996.2    0.07       0
  5000.2    0.16       0
Bank Sta=4996.2,5000.2
Exp/Cntr=0.3,0.1

Type RM Length L Ch R = 1,3964,78,78,78
BEGIN DESCRIPTION:
Elm 76 3963.78
END DESCRIPTION:
XS GIS Cut Line= 3
      1530522.02      6762098.28      1530541.55      6761940.70
      1530603.69      6761802.19
#Sta/Elev= 30
  4837.9 2168.86  4848.3 2166.97  4878.5 2156.59  4903.2 2152.61  4918.8 2147.92
  4949.0 2141.04  4959.1 2137.00  4966.7 2131.70  4969.2 2129.95  4984.2 2127.04
  4987.3 2124.95  4987.6 2124.45  4991.3 2124.95  4995.5 2126.49  5000.9 2126.49
  5010.6 2132.13  5016.7 2137.54  5022.2 2137.24  5032.5 2141.49  5054.4 2142.72
  5063.1 2145.61  5068.5 2144.93  5086.2 2151.77  5091.7 2150.68  5109.2 2157.47
  5114.9 2160.60  5120.4 2159.28  5138.1 2162.70  5143.6 2160.41  5148.5 2160.24
#Mann=4,-1,0
  4837.9    0.07       0  4966.7    0.16       0  4987.3    0.07       0
  4991.3    0.16       0
Bank Sta=4987.3,4991.3
Exp/Cntr=0.3,0.1

Type RM Length L Ch R = 1,3886,99,99,99
BEGIN DESCRIPTION:
Elm 76 3886.478
END DESCRIPTION:
XS GIS Cut Line= 3
      1530555.00      6762087.99      1530620.20      6761937.51
      1530654.99      6761888.01
#Sta/Elev= 30
  4836.0 2171.50  4838.7 2171.50  4845.0 2168.77  4850.5 2170.85  4868.5 2163.14
  4873.9 2162.27  4879.6 2158.08  4897.4 2150.29  4920.9 2142.84  4927.2 2140.25
  4934.1 2138.64  4944.4 2137.97  4955.9 2134.92  4966.8 2134.20  4973.3 2132.52
  4978.7 2132.32  4988.6 2125.37  4996.8 2125.23  4997.7 2124.20  4998.0 2123.70
  5001.5 2123.70  5001.7 2124.20  5002.8 2124.20  5017.4 2132.72  5023.8 2135.63
  5032.2 2137.91  5038.3 2140.57  5047.0 2140.86  5053.1 2143.95  5060.5 2144.79
#Mann=4,-1,0
  4836.0    0.07       0  4927.2    0.16       0  4997.7    0.07       0
  5001.7    0.16       0
Bank Sta=4997.7,5001.7
Exp/Cntr=0.3,0.1

Type RM Length L Ch R = 1,3787,76,76,76
BEGIN DESCRIPTION:
Elm 76 3786.89
END DESCRIPTION:
XS GIS Cut Line= 3
      1530626.18      6762113.88      1530696.50      6761996.69
      1530768.13      6761863.84
#Sta/Elev= 30
  4850.7 2172.50  4854.9 2171.90  4860.8 2173.05  4869.2 2172.78  4882.1 2170.83
  4891.9 2168.35  4897.7 2165.47  4904.2 2160.17  4919.1 2150.33  4936.5 2141.56
  4956.0 2132.59  4962.5 2127.89  4975.4 2123.28  4975.6 2122.78  4979.4 2123.28
  4993.2 2123.77  4998.8 2129.39  5008.6 2136.45  5015.1 2139.85  5020.7 2139.65
  5031.3 2141.61  5053.2 2143.64  5058.8 2145.16  5075.1 2146.22  5080.7 2147.72
  5088.1 2147.87  5097.0 2149.79  5102.6 2149.38  5118.9 2151.17  5138.3 2151.77
#Mann=4,-1,0
  4850.7    0.07       0  4936.5    0.16       0  4975.4    0.07       0
  4979.4    0.16       0
Bank Sta=4975.4,4979.4
Exp/Cntr=0.3,0.1

Type RM Length L Ch R = 1,3711,93,93,93
BEGIN DESCRIPTION:
Elm 76 3711.36
END DESCRIPTION:
XS GIS Cut Line= 3
      1530686.07      6762130.82      1530759.00      6762034.45
      1530850.09      6761857.47
#Sta/Elev= 30
  4878.7 2173.00  4901.4 2170.83  4907.7 2167.97  4916.0 2166.11  4944.9 2152.89
  4951.4 2146.90  4965.9 2137.71  4972.2 2135.70  4980.5 2131.03  4986.7 2129.78
  4994.2 2123.56  5003.4 2121.35  5005.1 2120.89  5005.3 2120.39  5008.8 2120.39
  5009.1 2120.89  5018.0 2122.13  5023.6 2121.05  5029.3 2126.56  5045.8 2137.16
  5051.8 2139.80  5062.4 2140.97  5074.3 2143.69  5090.2 2144.56  5128.9 2148.58
  5134.5 2148.52  5141.8 2149.85  5156.7 2150.66  5171.8 2152.18  5198.6 2154.65
#Mann=5,-1,0
  4878.7    0.07       0  5003.4    0.16       0  5005.1    0.07       0
  5009.1    0.16       0  5171.8    0.07       0
Bank Sta=5005.1,5009.1
Exp/Cntr=0.3,0.1

Type RM Length L Ch R = 1,3618,71,71,71
BEGIN DESCRIPTION:
Elm 76 3618.22
END DESCRIPTION:
XS GIS Cut Line= 3
      1530735.53      6762142.55      1530851.45      6762042.26
      1530945.18      6761883.44
#Sta/Elev= 30
  4847.0 2171.58  4885.8 2171.11  4892.4 2165.11  4899.2 2164.78  4906.6 2167.90
  4913.9 2160.23  4920.9 2160.85  4927.5 2152.44  4935.1 2151.46  4941.7 2144.80
  4949.4 2141.11  4956.0 2131.50  4963.6 2129.48  4970.3 2124.68  4977.9 2124.15
  4989.8 2119.56  4990.0 2119.06  4993.8 2119.56  5005.7 2120.26  5014.1 2127.17
  5019.9 2129.22  5028.5 2135.45  5051.2 2139.25  5057.0 2138.29  5072.6 2144.83
  5130.0 2145.06  5144.6 2147.30  5152.6 2153.27  5174.1 2156.78  5184.7 2156.61
#Mann=5,-1,0
  4847.0    0.07       0  4913.9    0.16       0  4989.8    0.07       0
  4993.8    0.16       0  5130.0    0.07       0
Bank Sta=4989.8,4993.8
Exp/Cntr=0.3,0.1

Type RM Length L Ch R = 1,3547,66,66,66
BEGIN DESCRIPTION:
Elm 76 3547.33
END DESCRIPTION:
XS GIS Cut Line= 3
      1530762.94      6762138.60      1530908.74      6762086.53
      1531018.09      6761936.83
#Sta/Elev= 30
  4849.9 2170.67  4867.3 2170.70  4885.6 2168.01  4892.8 2165.09  4898.1 2164.94
  4905.2 2159.11  4937.0 2143.25  4979.5 2133.92  4990.5 2127.02  5000.1 2122.98
  5004.7 2122.98  5008.0 2121.08  5020.6 2118.46  5020.9 2117.96  5024.6 2118.46
  5037.3 2122.26  5043.5 2127.44  5052.0 2129.77  5058.2 2128.98  5072.8 2135.58
  5079.0 2135.17  5087.5 2138.02  5093.7 2137.40  5108.4 2144.19  5114.6 2139.23
  5123.0 2140.61  5129.2 2137.94  5142.3 2141.64  5158.6 2146.84  5190.1 2149.94
#Mann=5,-1,0
  4849.9    0.07       0  4885.6    0.16       0  5020.6    0.07       0
  5024.6    0.16       0  5142.3    0.07       0
Bank Sta=5020.6,5024.6
Exp/Cntr=0.3,0.1

Type RM Length L Ch R = 1,3481,84,84,84
BEGIN DESCRIPTION:
Elm 76 3480.74
END DESCRIPTION:
XS GIS Cut Line= 3
      1530756.37      6762162.05      1530949.10      6762137.31
      1531111.54      6762133.44
#Sta/Elev= 30
  4807.6 2169.34  4836.5 2167.81  4846.5 2166.31  4859.0 2161.36  4866.7 2157.69
  4875.2 2152.51  4880.3 2154.07  4886.9 2148.55  4897.0 2143.35  4907.0 2139.95
  4917.1 2137.96  4947.4 2136.36  4954.8 2133.56  4959.9 2133.41  4967.5 2129.24
  4977.6 2125.55  4987.7 2119.80  4995.3 2117.95  4995.6 2117.45  4999.1 2117.45
  4999.3 2117.95  5007.8 2119.41  5027.8 2125.29  5047.8 2129.03  5067.8 2141.04
  5077.8 2143.65  5096.3 2149.84  5117.8 2154.42  5137.8 2156.69  5164.4 2158.29
#Mann=5,-1,0
  4807.6    0.07       0  4859.0    0.16       0  4995.3    0.07       0
  4999.3    0.16       0  5096.3    0.07       0
Bank Sta=4995.3,4999.3
Exp/Cntr=0.3,0.1

Type RM Length L Ch R = 1,3397,80,80,80
BEGIN DESCRIPTION:
Elm 76 3397.37
END DESCRIPTION:
XS GIS Cut Line= 3
      1530734.31      6762195.91      1530902.23      6762207.62
      1531126.17      6762203.72
#Sta/Elev= 30
  4828.2 2169.11  4831.0 2169.11  4838.9 2166.97  4848.9 2166.29  4869.0 2157.80
  4879.0 2155.19  4899.1 2147.04  4909.1 2144.93  4919.0 2140.22  4927.1 2136.98
  4932.1 2139.37  4949.2 2132.54  4959.2 2129.39  4969.2 2128.29  4989.3 2124.26
  4995.4 2119.54  5000.4 2119.54  5007.3 2117.48  5007.6 2116.98  5011.3 2117.48
  5019.3 2119.15  5029.3 2122.80  5069.3 2133.92  5099.3 2139.66  5109.3 2143.63
  5126.9 2148.62  5139.3 2153.56  5149.3 2156.06  5199.3 2163.17  5220.5 2163.30
#Mann=5,-1,0
  4828.2    0.07       0  4919.0    0.16       0  5007.3    0.07       0
  5011.3    0.16       0  5126.9    0.07       0
Bank Sta=5007.3,5011.3
Exp/Cntr=0.3,0.1

Type RM Length L Ch R = 1,3317,85,85,85
BEGIN DESCRIPTION:
Elm 76 3317.1
END DESCRIPTION:
XS GIS Cut Line= 3
      1530721.28      6762244.09      1530867.07      6762275.33
      1531070.13      6762335.21
#Sta/Elev= 30
  4849.8 2171.05  4863.8 2170.57  4904.7 2167.53  4915.0 2165.72  4935.2 2155.54
  4940.3 2150.60  4945.6 2146.20  4955.9 2139.84  4966.1 2132.72  4982.5 2125.46
  4989.7 2122.44  4995.3 2119.02  5007.2 2117.89  5027.6 2116.83  5027.9 2116.33
  5031.4 2116.33  5031.6 2116.83  5038.4 2122.54  5048.9 2128.34  5057.7 2131.59
  5062.9 2134.51  5069.7 2136.35  5080.1 2137.06  5096.3 2139.40  5111.4 2139.19
  5153.2 2142.56  5162.9 2142.73  5194.8 2146.21  5206.6 2148.61  5210.6 2150.05
#Mann=5,-1,0
  4849.8    0.07       0  4982.5    0.16       0  5027.6    0.07       0
  5031.6    0.16       0  5153.2    0.07       0
Bank Sta=5027.6,5031.6
Exp/Cntr=0.3,0.1

Type RM Length L Ch R = 1,3232,104,104,104
BEGIN DESCRIPTION:
Elm 76 3232.28
END DESCRIPTION:
XS GIS Cut Line= 3
      1530708.20      6762336.53      1530855.35      6762357.36
      1531084.50      6762341.74
#Sta/Elev= 30
  4852.2 2167.75  4896.4 2167.29  4909.6 2166.18  4919.7 2164.56  4929.8 2160.39
  4939.9 2149.62  4950.0 2127.84  4960.1 2116.67  4970.5 2115.60  4970.7 2115.10
  4974.2 2115.10  4974.5 2115.60  4980.3 2117.40  4990.4 2119.42  4998.1 2120.05
  5020.5 2120.14  5027.9 2120.87  5040.6 2123.19  5050.6 2126.70  5060.3 2130.59
  5065.3 2131.59  5070.6 2133.62  5100.7 2136.58  5110.7 2136.98  5120.7 2138.18
  5156.6 2141.49  5180.9 2143.32  5190.9 2144.72  5221.0 2150.05  5230.5 2150.79
#Mann=5,-1,0
  4852.2    0.07       0  4970.5    0.07       0  4974.5    0.07       0
  5027.9    0.16       0  5156.6    0.07       0
Bank Sta=4970.5,4974.5
Exp/Cntr=0.3,0.1

Type RM Length L Ch R = 1,3128,85,85,85
BEGIN DESCRIPTION:
Elm 76 3127.6
END DESCRIPTION:
XS GIS Cut Line= 3
      1530717.36      6762482.36      1530876.19      6762456.32
      1531089.77      6762356.04
#Sta/Elev= 30
  4841.9 2161.40  4849.6 2157.82  4869.9 2151.70  4880.0 2150.29  4890.2 2152.86
  4902.6 2158.70  4920.6 2163.73  4940.8 2164.73  4958.8 2163.52  4963.9 2157.01
  4971.2 2123.37  4979.4 2114.98  4979.6 2114.48  4983.4 2114.98  5005.0 2116.89
  5008.9 2118.03  5044.1 2119.51  5054.5 2120.76  5077.3 2130.00  5082.8 2131.30
  5100.1 2132.40  5134.1 2138.00  5143.0 2138.09  5151.3 2137.75  5174.1 2139.52
  5196.9 2142.18  5202.4 2143.88  5219.7 2145.85  5233.4 2149.01  5238.8 2149.01
#Mann=5,-1,0
  4841.9    0.07       0  4979.4    0.07       0  4983.4    0.07       0
  5044.1    0.16       0  5143.0    0.07       0
Bank Sta=4979.4,4983.4
Exp/Cntr=0.3,0.1

Type RM Length L Ch R = 1,3043,160,160,160
BEGIN DESCRIPTION:
Elm 76 3042.76
END DESCRIPTION:
XS GIS Cut Line= 3
      1530735.55      6762574.81      1530932.18      6762517.52
      1531100.14      6762383.15
#Sta/Elev= 30
  4792.9 2155.11  4795.2 2155.11  4798.5 2151.76  4803.7 2152.83  4832.0 2146.23
  4837.2 2147.50  4854.8 2143.63  4870.7 2136.12  4904.2 2144.82  4909.4 2150.39
  4927.7 2154.03  4942.9 2159.56  4959.0 2140.23  4969.4 2122.18  4976.4 2115.47
  4994.6 2113.90  4994.8 2113.40  4998.6 2113.90  5008.4 2114.63  5027.1 2118.48
  5056.0 2128.42  5078.2 2123.99  5084.8 2124.40  5113.6 2128.99  5120.0 2133.51
  5134.4 2136.22  5169.6 2139.11  5192.0 2143.36  5198.4 2142.04  5212.8 2146.49
#Mann=4,-1,0
  4792.9    0.07       0  4994.6    0.07       0  4998.6    0.07       0
  5008.4    0.16       0
Bank Sta=4994.6,4998.6
Exp/Cntr=0.3,0.1

Type RM Length L Ch R = 1,2883,89,89,89
BEGIN DESCRIPTION:
Elm 76 2883.2
END DESCRIPTION:
XS GIS Cut Line= 3
      1530873.61      6762712.81      1531080.61      6762548.77
      1531178.12      6762392.76
#Sta/Elev= 30
  4724.9 2151.14  4729.0 2151.14  4736.9 2147.97  4743.3 2148.25  4751.3 2145.70
  4757.7 2145.68  4772.1 2140.88  4778.5 2140.89  4792.9 2138.85  4865.2 2132.92
  4921.1 2126.30  4929.2 2123.08  4935.6 2123.18  4950.0 2118.20  4985.2 2114.03
  4988.6 2112.73  5020.5 2112.50  5020.8 2112.00  5024.5 2112.50  5028.4 2112.89
  5037.1 2118.11  5049.6 2134.25  5059.1 2139.22  5065.0 2141.36  5080.3 2143.14
  5101.5 2144.21  5116.8 2146.70  5144.0 2149.24  5159.3 2151.23  5173.0 2154.38
#Mann=4,-1,0
  4724.9    0.07       0  4865.2    0.16       0  5020.5    0.07       0
  5024.5    0.16       0
Bank Sta=5020.5,5024.5
Exp/Cntr=0.3,0.1

Type RM Length L Ch R = 1,2794,99,99,99
BEGIN DESCRIPTION:
Elm 76 2794.08
END DESCRIPTION:
XS GIS Cut Line= 3
      1530910.05      6762744.08      1531131.40      6762608.67
      1531296.75      6762503.20
#Sta/Elev= 30
  4743.8 2151.61  4750.7 2146.35  4760.2 2144.09  4766.1 2141.33  4781.5 2136.68
  4787.4 2136.70  4802.9 2134.52  4839.6 2134.32  4856.2 2136.59  4876.3 2135.97
  4882.2 2133.00  4897.6 2135.81  4903.5 2130.28  4913.1 2128.84  4919.0 2126.69
  4925.4 2125.54  4940.3 2124.78  4948.9 2123.00  4955.7 2120.39  4984.1 2112.51
  5011.6 2111.27  5011.9 2110.77  5015.6 2111.27  5019.6 2111.44  5028.9 2116.77
  5034.8 2119.36  5043.1 2124.82  5050.0 2126.13  5114.3 2131.97  5199.4 2137.98
#Mann=4,-1,0
  4743.8    0.07       0  4856.2    0.16       0  5011.6    0.07       0
  5015.6    0.16       0
Bank Sta=5011.6,5015.6
Exp/Cntr=0.3,0.1

Type RM Length L Ch R = 1,2695,84,84,84
BEGIN DESCRIPTION:
Elm 76 2695.11
END DESCRIPTION:
XS GIS Cut Line= 3
      1530986.90      6762810.47      1531205.61      6762676.37
      1531312.70      6762521.55
#Sta/Elev= 30
  4752.7 2147.14  4761.7 2145.43  4767.5 2141.67  4773.9 2139.67  4810.1 2130.60
  4832.6 2125.84  4838.9 2126.37  4841.0 2126.54  4846.8 2123.05  4856.0 2123.05
  4862.3 2119.91  4868.1 2124.05  4877.7 2122.59  4883.6 2128.21  4899.0 2118.39
  4904.9 2119.87  4914.4 2115.58  4941.6 2114.64  4972.5 2110.99  5004.0 2110.20
  5004.2 2109.70  5008.0 2110.20  5030.0 2111.04  5036.1 2112.25  5043.7 2121.70
  5051.0 2126.83  5065.8 2127.58  5092.9 2131.04  5137.5 2133.19  5197.5 2137.75
#Mann=4,-1,0
  4752.7    0.07       0  4838.9    0.16       0  5004.0    0.07       0
  5008.0    0.16       0
Bank Sta=5004,5008
Exp/Cntr=0.3,0.1

Type RM Length L Ch R = 1,2611,93,93,93
BEGIN DESCRIPTION:
Elm 76 2611.37
END DESCRIPTION:
XS GIS Cut Line= 3
      1531005.08      6762832.63      1531255.09      6762742.78
      1531391.53      6762687.43
#Sta/Elev= 30
  4738.3 2150.84  4765.8 2147.09  4771.1 2142.22  4791.2 2140.90  4796.5 2135.66
  4812.6 2129.22  4817.0 2126.23  4821.9 2122.90  4833.9 2117.54  4852.6 2115.08
  4888.7 2114.66  4929.5 2111.27  4944.8 2111.37  4961.4 2109.05  4980.6 2108.67
  4980.9 2108.17  4984.6 2108.67  5036.2 2110.23  5047.0 2114.87  5054.5 2125.85
  5059.9 2129.34  5068.6 2132.19  5084.0 2135.07  5101.0 2140.03  5108.1 2143.17
  5122.6 2145.40  5132.2 2145.65  5137.9 2147.37  5144.2 2148.49  5151.2 2152.35
#Mann=5,-1,0
  4738.3    0.07       0  4817.0    0.16       0  4980.6    0.07       0
  4984.6    0.16       0  5137.9    0.07       0
Bank Sta=4980.6,4984.6
Exp/Cntr=0.3,0.1

Type RM Length L Ch R = 1,2518,77,77,77
BEGIN DESCRIPTION:
Elm 76 2518.43
END DESCRIPTION:
XS GIS Cut Line= 3
      1531055.87      6762905.54      1531261.60      6762835.23
      1531420.91      6762751.04
#Sta/Elev= 30
  4784.8 2154.77  4796.2 2154.58  4815.6 2150.72  4822.2 2147.74  4836.7 2137.68
  4853.5 2123.37  4862.4 2118.59  4879.0 2114.01  4884.8 2110.54  4890.1 2111.31
  4921.4 2108.60  4953.0 2111.88  4973.5 2108.68  5015.4 2107.72  5015.6 2107.22
  5019.4 2107.72  5053.4 2108.63  5069.7 2113.19  5075.4 2117.30  5085.2 2117.93
  5091.7 2121.94  5107.9 2126.75  5113.8 2131.56  5132.6 2134.04  5135.8 2133.87
  5152.1 2138.70  5157.8 2138.18  5174.1 2144.96  5179.8 2143.73  5182.4 2147.25
#Mann=5,-1,0
  4784.8    0.07       0  4862.4    0.16       0  5015.4    0.07       0
  5019.4    0.16       0  5132.6    0.07       0
Bank Sta=5015.4,5019.4
Exp/Cntr=0.3,0.1

Type RM Length L Ch R = 1,2441,78,78,78
BEGIN DESCRIPTION:
Elm 76 2440.941
END DESCRIPTION:
XS GIS Cut Line= 3
      1531104.99      6762988.01      1531303.77      6762898.51
      1531455.00      6762788.00
#Sta/Elev= 30
  4782.0 2151.29  4796.3 2150.10  4819.5 2145.31  4836.8 2139.39  4848.1 2134.04
  4857.5 2131.93  4865.8 2131.37  4871.3 2125.55  4888.9 2126.03  4894.4 2116.63
  4912.1 2116.61  4917.5 2111.69  4935.2 2113.12  5006.5 2105.81  5006.8 2105.31
  5010.5 2105.81  5014.7 2107.05  5064.9 2107.76  5088.1 2113.89  5108.9 2120.95
  5115.1 2124.92  5123.6 2134.71  5129.8 2140.37  5137.8 2145.39  5144.4 2151.44
  5159.1 2160.34  5173.8 2165.51  5180.0 2162.79  5184.2 2165.69  5187.3 2165.69
#Mann=4,-1,0
  4782.0    0.07       0  4857.5    0.16       0  5006.5    0.07       0
  5010.5    0.16       0
Bank Sta=5006.5,5010.5
Exp/Cntr=0.3,0.1

Type RM Length L Ch R = 1,2363,76,76,76
BEGIN DESCRIPTION:
Elm 76 2362.67
END DESCRIPTION:
XS GIS Cut Line= 3
      1531127.51      6763035.74      1531312.38      6762974.55
      1531506.37      6762888.62
#Sta/Elev= 30
  4812.3 2148.61  4823.2 2148.90  4830.7 2147.51  4849.7 2141.42  4859.2 2139.74
  4904.5 2125.91  4913.1 2124.18  4918.4 2125.42  4950.1 2121.62  4957.1 2119.74
  4967.7 2115.22  4976.5 2108.35  4981.8 2109.42  4986.7 2104.94  4987.0 2104.44
  4990.7 2104.94  5059.7 2105.69  5088.4 2109.31  5111.7 2118.15  5129.5 2127.55
  5135.0 2129.27  5141.1 2136.06  5158.3 2143.95  5174.0 2148.90  5181.6 2153.02
  5187.0 2151.75  5204.8 2158.93  5210.3 2158.57  5215.7 2161.53  5219.2 2161.53
#Mann=4,-1,0
  4812.3    0.07       0  4859.2    0.16       0  4986.7    0.07       0
  4990.7    0.16       0
Bank Sta=4986.7,4990.7
Exp/Cntr=0.3,0.1

Type RM Length L Ch R = 1,2287,114,114,114
BEGIN DESCRIPTION:
Elm 76 2287.29
END DESCRIPTION:
XS GIS Cut Line= 3
      1531157.48      6763104.75      1531318.90      6763048.77
      1531518.15      6762944.58
#Sta/Elev= 30
  4830.9 2136.75  4834.9 2135.04  4840.2 2131.24  4849.4 2127.82  4860.0 2125.91
  4866.0 2122.84  4871.3 2126.52  4891.8 2122.78  4897.2 2120.97  4902.5 2121.41
  4909.0 2120.54  4923.0 2118.32  4928.3 2118.53  4959.4 2115.20  4985.3 2105.55
  4995.0 2104.56  4995.3 2104.06  4999.0 2104.56  5036.3 2105.46  5119.0 2104.66
  5155.3 2110.71  5163.1 2112.49  5168.8 2115.23  5177.9 2117.18  5185.2 2122.16
  5190.8 2132.76  5200.5 2140.69  5212.9 2150.03  5222.0 2154.28  5226.6 2154.28
#Mann=4,-1,0
  4830.9   0.035       0  4909.0    0.16       0  4995.0    0.07       0
  4999.0    0.16       0
Bank Sta=4995,4999
Exp/Cntr=0.3,0.1

Type RM Length L Ch R = 1,2173,80,80,80
BEGIN DESCRIPTION:
Elm 76 2172.92
END DESCRIPTION:
XS GIS Cut Line= 3
      1531208.18      6763152.94      1531391.81      6763133.40
      1531580.28      6763071.01
#Sta/Elev= 30
  4811.0 2125.65  4817.9 2123.55  4838.0 2120.01  4848.0 2119.43  4870.6 2115.95
  4888.3 2114.19  4898.3 2112.29  4904.2 2110.32  4909.2 2110.48  4918.4 2107.38
  4928.5 2106.42  4968.7 2104.15  5000.6 2104.07  5025.1 2102.84  5025.3 2102.34
  5028.8 2102.34  5029.1 2102.84  5041.2 2102.91  5051.7 2104.20  5058.8 2106.73
  5064.0 2105.31  5083.3 2109.04  5090.5 2111.29  5095.8 2108.65  5122.2 2119.75
  5127.5 2119.58  5178.1 2135.82  5185.6 2141.25  5190.9 2142.71  5194.2 2147.27
#Mann=4,-1,0
  4811.0   0.035       0  4870.6    0.16       0  5025.1    0.07       0
  5029.1    0.16       0
Bank Sta=5025.1,5029.1
Exp/Cntr=0.3,0.1

Type RM Length L Ch R = 1,2093,123,123,123
BEGIN DESCRIPTION:
Elm 76 2092.81
END DESCRIPTION:
XS GIS Cut Line= 3
      1531223.82      6763267.53      1531402.23      6763211.53
      1531597.58      6763106.04
#Sta/Elev= 30
  4809.8 2123.11  4820.6 2123.12  4825.8 2122.29  4832.0 2118.37  4852.3 2113.59
  4863.5 2112.38  4873.9 2110.47  4884.4 2108.15  4890.7 2105.80  4895.9 2105.68
  4923.1 2102.22  4945.3 2101.70  4945.5 2101.20  4949.0 2101.20  4949.3 2101.70
  5015.9 2102.59  5032.1 2102.28  5056.4 2103.65  5090.9 2107.92  5103.4 2110.59
  5135.8 2114.79  5157.7 2121.59  5163.4 2122.09  5170.4 2125.85  5179.6 2129.65
  5185.3 2130.64  5193.1 2134.87  5201.5 2138.32  5214.5 2144.93  5218.8 2144.93
#Mann=5,-1,0
  4809.8   0.035       0  4852.3    0.07       0  4945.3    0.07       0
  4949.3    0.07       0  5056.4    0.16       0
Bank Sta=4945.3,4949.3
Exp/Cntr=0.3,0.1

Type RM Length L Ch R = 1,1970,136,136,136
BEGIN DESCRIPTION:
Elm 76 1969.96
END DESCRIPTION:
XS GIS Cut Line= 3
      1531239.44      6763372.99      1531407.44      6763332.62
      1531601.36      6763145.16
#Sta/Elev= 30
  4827.5 2117.14  4833.2 2118.24  4849.9 2114.82  4874.9 2111.45  4911.7 2102.89
  4953.7 2099.41  4985.5 2098.28  4985.7 2097.78  4989.5 2098.28  5023.1 2098.71
  5037.3 2099.98  5044.2 2099.67  5051.4 2100.98  5072.5 2099.89  5100.8 2100.06
  5108.0 2101.10  5178.5 2102.15  5185.7 2102.57  5199.9 2106.20  5206.8 2109.79
  5211.2 2110.84  5214.0 2111.50  5221.0 2116.66  5228.2 2115.77  5235.1 2120.47
  5242.3 2119.38  5249.3 2124.02  5256.5 2123.79  5263.4 2132.09  5270.0 2132.08
#Mann=5,-1,0
  4827.5   0.035       0  4849.9    0.07       0  4985.5    0.07       0
  4989.5    0.07       0  5211.2    0.16       0
Bank Sta=4985.5,4989.5
Exp/Cntr=0.3,0.1

Type RM Length L Ch R = 1,1834,66,66,66
BEGIN DESCRIPTION:
Elm 76 1833.68
END DESCRIPTION:
XS GIS Cut Line= 3
      1531182.13      6763396.42      1531416.55      6763434.19
      1531681.77      6763524.75
#Sta/Elev= 30
  4766.8 2119.00  4820.4 2114.01  4830.5 2114.96  4845.7 2113.70  4868.5 2111.30
  4901.4 2105.05  4930.3 2104.30  4935.4 2101.78  4992.1 2100.12  4997.2 2097.05
  5000.9 2096.61  5013.2 2096.37  5030.3 2098.21  5033.4 2093.92  5033.7 2093.42
  5037.8 2093.92  5055.4 2095.29  5061.6 2097.00  5066.9 2094.67  5092.9 2099.63
  5098.2 2097.58  5124.2 2098.40  5129.5 2097.41  5150.3 2099.72  5161.1 2098.41
  5186.9 2100.21  5218.2 2105.24  5224.5 2108.43  5256.2 2116.00  5284.5 2120.70
#Mann=4,-1,0
  4766.8   0.035       0  4845.7    0.07       0  5033.4    0.07       0
  5037.8    0.07       0
Bank Sta=5033.4,5037.8
Exp/Cntr=0.3,0.1

Type RM Length L Ch R = 1,1768,93,93,93
BEGIN DESCRIPTION:
Elm 76 1768.38
END DESCRIPTION:
XS GIS Cut Line= 3
      1531209.50      6763522.73      1531402.23      6763496.69
      1531660.68      6763552.53
#Sta/Elev= 30
  4802.7 2116.89  4808.3 2115.19  4828.4 2111.78  4889.0 2105.71  4939.4 2098.40
  4952.3 2098.86  4959.0 2094.38  4969.7 2094.19  4979.8 2092.86  4989.9 2093.49
  5001.2 2092.68  5008.0 2088.34  5008.3 2087.84  5012.1 2087.84  5012.4 2088.34
  5031.5 2090.45  5070.5 2092.29  5075.6 2093.88  5081.9 2094.70  5112.6 2096.44
  5119.7 2098.78  5124.8 2096.57  5143.2 2097.43  5163.7 2099.71  5169.0 2101.21
  5204.6 2104.92  5218.2 2107.54  5235.3 2112.26  5255.8 2118.31  5261.6 2121.08
#Mann=4,-1,0
  4802.7    0.16       0  4959.0    0.07       0  5008.0    0.07       0
  5012.4    0.07       0
Bank Sta=5008,5012.4
Exp/Cntr=0.3,0.1

Type RM Length L Ch R = 1,1675,78,78,78
BEGIN DESCRIPTION:
Elm 76 1675.45
END DESCRIPTION:
XS GIS Cut Line= 3
      1531193.93      6763572.21      1531399.62      6763589.13
      1531615.74      6763598.25
#Sta/Elev= 30
  4794.4 2118.81  4802.3 2118.68  4807.3 2116.83  4855.7 2114.91  4865.7 2113.66
  4885.8 2109.33  4905.8 2106.40  4915.9 2103.85  4928.5 2098.97  4935.9 2096.79
  4956.0 2094.67  4966.0 2092.50  4976.1 2089.15  4983.9 2087.33  4984.2 2086.83
  4988.0 2086.83  4988.3 2087.33  4996.0 2088.42  5026.2 2090.23  5036.2 2091.31
  5046.2 2093.28  5065.6 2094.85  5091.9 2095.90  5116.3 2097.60  5126.3 2098.98
  5166.3 2102.80  5176.3 2105.19  5206.3 2109.56  5214.2 2111.35  5217.1 2111.35
#Mann=4,-1,0
  4794.4    0.16       0  4983.9    0.07       0  4988.3    0.16       0
  5065.6    0.07       0
Bank Sta=4983.9,4988.3
Exp/Cntr=0.3,0.1

Type RM Length L Ch R = 1,1597,84,84,84
BEGIN DESCRIPTION:
Elm 76 1597.08
END DESCRIPTION:
XS GIS Cut Line= 3
      1531174.41      6763633.41      1531354.05      6763652.94
      1531600.03      6763663.35
#Sta/Elev= 30
  4816.7 2118.34  4819.5 2118.34  4839.3 2114.12  4857.5 2110.31  4877.6 2107.37
  4897.8 2105.70  4904.1 2104.40  4938.0 2100.81  4968.2 2095.47  4978.2 2095.04
  4995.4 2092.27  5001.1 2091.94  5006.2 2086.90  5006.5 2086.40  5010.3 2086.40
  5010.6 2086.90  5018.4 2087.51  5028.4 2090.36  5058.4 2092.50  5068.4 2092.28
  5078.4 2093.28  5088.4 2093.22  5118.5 2097.69  5152.3 2100.30  5178.5 2103.89
  5208.5 2109.39  5218.5 2110.56  5228.6 2112.54  5239.5 2115.94  5243.6 2116.30
#Mann=5,-1,0
  4816.7    0.07       0  4839.3    0.16       0  5006.2    0.07       0
  5010.6    0.16       0  5152.3    0.07       0
Bank Sta=5006.2,5010.6
Exp/Cntr=0.3,0.1

Type RM Length L Ch R = 1,1513,62,62,62
BEGIN DESCRIPTION:
Elm 76 1513.36
END DESCRIPTION:
XS GIS Cut Line= 3
      1531152.25      6763742.78      1531385.30      6763724.55
      1531589.71      6763688.10
#Sta/Elev= 30
  4760.4 2126.05  4764.3 2126.05  4783.2 2122.17  4813.3 2115.28  4828.1 2110.67
  4853.4 2104.89  4873.5 2103.02  4882.2 2101.37  4887.2 2101.86  4933.7 2094.84
  4963.8 2092.74  4973.8 2089.50  4981.6 2085.78  4981.9 2085.28  4985.7 2085.28
  4986.0 2085.78  5014.2 2087.37  5024.3 2086.75  5034.5 2089.72  5085.3 2096.54
  5113.8 2103.02  5118.9 2101.38  5125.9 2103.29  5136.1 2104.59  5145.3 2106.91
  5166.5 2111.61  5172.7 2114.07  5177.8 2113.54  5196.9 2116.02  5201.8 2116.02
#Mann=5,-1,0
  4760.4    0.07       0  4828.1    0.16       0  4981.6    0.07       0
  4986.0    0.16       0  5145.3    0.07       0
Bank Sta=4981.6,4986
Exp/Cntr=0.3,0.1

Type RM Length L Ch R = 1,1451,55,55,55
BEGIN DESCRIPTION:
Elm 76 1450.65
END DESCRIPTION:
XS GIS Cut Line= 3
      1531155.01      6763838.00      1531435.38      6763767.88
      1531555.00      6763738.00
#Sta/Elev= 30
  4711.0 2140.25  4734.2 2138.47  4762.5 2123.14  4770.2 2117.53  4775.4 2118.48
  4783.1 2113.30  4796.2 2108.42  4811.5 2103.04  4816.6 2105.38  4845.0 2097.20
  4852.7 2094.21  4857.9 2096.14  4865.6 2093.76  4875.9 2091.73  4940.3 2091.75
  4948.1 2091.21  4958.4 2089.84  4979.3 2084.71  4979.6 2084.21  4983.7 2084.71
  4989.3 2086.26  5002.4 2086.70  5022.8 2091.85  5051.1 2095.59  5058.9 2098.23
  5064.0 2099.16  5092.4 2110.20  5100.1 2114.00  5113.0 2115.82  5123.3 2115.83
#Mann=4,-1,0
  4711.0    0.07       0  4796.2    0.16       0  4979.3    0.07       0
  4983.7    0.16       0
Bank Sta=4979.3,4983.7
Exp/Cntr=0.3,0.1

Type RM Length L Ch R = 1,1396,59,59,59
BEGIN DESCRIPTION:
Elm 76 1395.89
END DESCRIPTION:
XS GIS Cut Line= 3
      1531193.94      6763839.13      1531455.61      6763817.00
      1531648.35      6763809.19
#Sta/Elev= 30
  4737.9 2128.81  4740.9 2128.81  4749.0 2122.54  4759.0 2116.50  4785.8 2103.30
  4807.4 2096.27  4812.4 2098.09  4839.3 2090.97  4849.4 2089.46  4859.4 2088.83
  4869.4 2090.15  4899.5 2090.87  4919.6 2090.38  4927.0 2089.16  4969.8 2089.59
  4989.9 2086.02  4995.5 2084.22  4995.8 2083.72  4999.9 2084.22  5009.9 2085.07
  5029.9 2084.32  5039.9 2089.58  5059.9 2106.44  5080.0 2111.81  5090.0 2113.40
  5097.1 2112.48  5102.1 2113.35  5120.0 2112.19  5153.2 2113.66  5193.4 2115.22
#Mann=5,-1,0
  4737.9    0.07       0  4785.8    0.16       0  4995.5    0.07       0
  4999.9    0.16       0  5153.2    0.07       0
Bank Sta=4995.5,4999.9
Exp/Cntr=0.3,0.1

Type RM Length L Ch R = 1,1337,162,162,162
BEGIN DESCRIPTION:
Elm 76 1337.31
END DESCRIPTION:
XS GIS Cut Line= 3
      1531184.78      6763848.25      1531454.31      6763875.59
      1531628.83      6763952.43
#Sta/Elev= 30
  4729.8 2134.29  4732.4 2134.29  4740.1 2127.67  4770.2 2109.62  4776.1 2104.46
  4791.4 2099.00  4810.4 2093.86  4850.6 2086.92  4870.7 2089.71  4890.8 2089.72
  4900.9 2083.83  4908.7 2081.77  4909.0 2081.27  4913.1 2081.77  4941.1 2081.89
  5012.4 2085.73  5018.5 2086.57  5023.9 2090.39  5047.3 2092.29  5056.1 2095.50
  5065.1 2100.85  5070.6 2099.03  5077.9 2102.27  5093.9 2101.11  5110.7 2101.77
  5117.3 2103.47  5122.7 2102.20  5136.5 2104.84  5163.9 2109.80  5191.4 2111.40
#Mann=5,-1,0
  4729.8    0.07       0  4791.4    0.16       0  4908.7    0.07       0
  4913.1    0.16       0  5136.5    0.07       0
Bank Sta=4908.7,4913.1
Exp/Cntr=0.3,0.1

Type RM Length L Ch R = 1,1175,76,76,76
BEGIN DESCRIPTION:
Elm 76 1175.13
END DESCRIPTION:
XS GIS Cut Line= 3
      1531178.25      6763865.17      1531355.35      6763955.02
      1531584.50      6763996.68
#Sta/Elev= 30
  4801.9 2137.80  4817.1 2125.28  4822.8 2123.39  4839.4 2110.82  4845.0 2109.16
  4861.7 2098.91  4867.3 2098.01  4883.9 2092.10  4890.8 2091.04  4921.6 2085.29
  4944.0 2088.96  4988.9 2089.46  4995.3 2086.82  5002.9 2087.22  5010.3 2083.08
  5018.3 2081.12  5018.6 2080.62  5022.7 2081.12  5040.4 2085.93  5045.5 2085.75
  5051.0 2090.67  5061.1 2093.75  5098.9 2100.30  5103.9 2099.40  5111.9 2100.33
  5142.4 2098.00  5157.3 2098.29  5162.8 2099.83  5201.9 2103.91  5233.4 2107.51
#Mann=5,-1,0
  4801.9    0.07       0  4890.8    0.16       0  5018.3    0.07       0
  5022.7    0.16       0  5201.9    0.07       0
Bank Sta=5018.3,5022.7
Exp/Cntr=0.3,0.1

Type RM Length L Ch R = 1,1099,120,120,120
BEGIN DESCRIPTION:
Elm 76 1099.1
END DESCRIPTION:
XS GIS Cut Line= 3
      1531150.90      6763915.94      1531341.03      6764030.54
      1531570.78      6764035.73
#Sta/Elev= 30
  4799.1 2134.06  4804.4 2134.06  4826.8 2121.41  4832.6 2119.48  4838.9 2114.96
  4848.1 2110.26  4854.0 2108.82  4869.5 2099.96  4875.3 2098.53  4885.0 2094.85
  4890.9 2093.62  4897.3 2091.11  4912.2 2087.83  4920.6 2086.71  4927.7 2084.62
  4946.3 2084.02  4964.6 2085.90  5014.1 2086.01  5025.6 2085.58  5035.1 2083.89
  5042.9 2081.09  5043.2 2080.59  5047.3 2081.09  5065.1 2085.16  5085.1 2086.97
  5095.1 2088.97  5105.1 2092.81  5167.2 2097.54  5235.1 2103.49  5250.9 2106.17
#Mann=5,-1,0
  4799.1    0.07       0  4946.3    0.16       0  5042.9    0.07       0
  5047.3    0.16       0  5167.2    0.07       0
Bank Sta=5042.9,5047.3
Exp/Cntr=0.3,0.1

Type RM Length L Ch R = 1,979,119,119,119
BEGIN DESCRIPTION:
Elm 76 978.72
END DESCRIPTION:
XS GIS Cut Line= 3
      1531100.17      6763960.25      1531245.98      6764072.21
      1531550.29      6764112.52
#Sta/Elev= 30
  4862.1 2141.36  4885.1 2138.90  4893.3 2133.96  4899.6 2133.81  4906.0 2128.10
  4914.1 2122.91  4920.4 2121.06  4928.6 2114.52  4943.1 2106.70  4963.9 2095.83
  4978.5 2091.56  4993.0 2084.36  4999.3 2079.55  5004.6 2077.44  5005.0 2076.94
  5009.1 2077.44  5034.6 2081.67  5051.0 2081.46  5085.3 2084.84  5095.4 2083.56
  5105.5 2080.03  5115.6 2078.73  5131.2 2079.26  5155.9 2083.92  5166.0 2087.78
  5186.2 2090.42  5196.3 2093.33  5240.3 2094.52  5307.2 2097.09  5352.9 2102.31
#Mann=5,-1,0
  4862.1    0.07       0  5004.6    0.07       0  5009.1    0.07       0
  5131.2    0.16       0  5240.3    0.07       0
Bank Sta=5004.6,5009.1
Exp/Cntr=0.3,0.1

Type RM Length L Ch R = 1,860,149,149,149
BEGIN DESCRIPTION:
Elm 76 859.97
END DESCRIPTION:
XS GIS Cut Line= 3
      1531036.37      6764094.35      1531201.71      6764162.05
      1531560.51      6764177.65
#Sta/Elev= 30
  4818.6 2141.00  4837.4 2144.14  4842.8 2141.98  4860.3 2142.70  4866.8 2141.46
  4872.2 2137.53  4890.8 2131.80  4903.6 2123.43  4914.4 2118.92  4920.2 2112.97
  4925.6 2111.85  4936.0 2107.26  4944.2 2100.02  4949.6 2100.27  4957.6 2095.42
  4973.6 2089.72  4981.5 2085.42  4996.3 2079.22  5001.4 2079.22  5008.3 2077.25
  5008.7 2076.75  5012.8 2077.25  5030.6 2077.91  5060.6 2083.60  5100.6 2086.18
  5140.7 2091.16  5230.8 2093.60  5260.8 2093.20  5300.8 2095.62  5356.4 2101.20
#Mann=4,-1,0
  4818.6    0.07       0  4981.5    0.16       0  5008.3    0.07       0
  5012.8    0.16       0
Bank Sta=5008.3,5012.8
Exp/Cntr=0.3,0.1

Type RM Length L Ch R = 1,711,151,151,151
BEGIN DESCRIPTION:
Elm 76 711.29
END DESCRIPTION:
XS GIS Cut Line= 3
      1531024.62      6764182.88      1531158.74      6764296.17
      1531450.84      6764320.83
#Sta/Elev= 30
  4825.4 2117.48  4829.0 2113.16  4836.8 2112.18  4843.3 2106.60  4851.1 2105.88
  4857.6 2102.22  4881.4 2098.00  4886.2 2097.80  4900.5 2094.93  4907.0 2094.61
  4914.8 2092.52  4921.3 2092.45  4929.1 2090.77  4949.9 2089.02  4964.2 2086.80
  4970.7 2087.21  4978.5 2085.20  4985.0 2085.80  4992.8 2081.73  5001.0 2083.26
  5007.2 2077.61  5015.0 2074.54  5015.3 2074.04  5019.5 2074.54  5027.3 2076.39
  5077.3 2083.72  5127.7 2084.27  5177.8 2088.73  5268.2 2091.29  5294.1 2093.13
#Mann=4,-1,0
  4825.4    0.07       0  4881.4    0.16       0  5015.0    0.07       0
  5019.5    0.16       0
Bank Sta=5015,5019.5
Exp/Cntr=0.3,0.1

Type RM Length L Ch R = 1,560,72,72,72
BEGIN DESCRIPTION:
Elm 76 560.409
END DESCRIPTION:
XS GIS Cut Line= 3
      1531012.94      6764380.81      1531196.86      6764431.94
      1531505.00      6764488.00
#Sta/Elev= 30
  4809.1 2091.95  4812.8 2091.95  4816.9 2090.44  4832.0 2088.53  4851.1 2086.73
  4883.9 2085.75  4904.7 2084.16  4924.8 2081.43  4929.9 2081.32  4935.8 2079.02
  4946.2 2076.84  4956.6 2075.83  4985.4 2074.84  4985.7 2074.34  4989.9 2074.84
  5000.0 2075.46  5018.5 2081.06  5028.6 2080.29  5057.9 2082.56  5130.2 2085.41
  5181.1 2089.68  5201.4 2090.62  5221.7 2093.73  5228.1 2095.37  5232.5 2095.04
  5272.5 2104.23  5281.4 2105.50  5286.5 2104.92  5303.0 2107.08  5313.2 2106.60
#Mann=5,-1,0
  4809.1    0.07       0  4985.4    0.07       0  4989.9    0.07       0
  5018.5    0.16       0  5232.5    0.07       0
Bank Sta=4985.4,4989.9
Exp/Cntr=0.3,0.1

Type RM Length L Ch R = 1,488,84,84,84
BEGIN DESCRIPTION:
Elm 76 4380
END DESCRIPTION:
XS GIS Cut Line= 3
      1531031.09      6764402.91      1531204.63      6764503.34
      1531470.03      6764603.00
#Sta/Elev= 30
  4799.5 2089.40  4804.7 2090.52  4814.7 2088.49  4820.5 2090.31  4827.1 2088.21
  4836.3 2087.01  4842.0 2087.89  4857.8 2085.13  4885.1 2083.58  4895.1 2081.81
  4959.7 2080.54  4965.8 2079.72  4975.5 2074.12  4981.2 2075.50  4986.6 2071.29
  4986.9 2070.79  4991.1 2071.29  4997.0 2073.27  5002.9 2073.21  5011.1 2077.45
  5029.8 2080.68  5075.2 2083.37  5107.2 2087.31  5131.4 2089.15  5198.1 2093.84
  5214.0 2095.69  5235.4 2100.09  5267.4 2101.75  5278.1 2103.01  5283.5 2104.86
#Mann=5,-1,0
  4799.5    0.07       0  4986.6    0.07       0  4991.1    0.07       0
  5029.8    0.16       0  5131.4    0.07       0
Bank Sta=4986.6,4991.1
Exp/Cntr=0.3,0.1

Type RM Length L Ch R = 1,404,43,43,43
BEGIN DESCRIPTION:
Elm 76 4379
END DESCRIPTION:
XS GIS Cut Line= 3
      1531025.91      6764417.24      1531201.48      6764586.55
      1531365.75      6764658.14
#Sta/Elev= 30
  4756.1 2093.03  4791.4 2089.77  4826.6 2083.52  4848.0 2082.81  4876.3 2079.99
  4968.1 2078.48  4982.3 2076.07  4989.5 2072.14  4994.2 2071.51  4994.5 2071.01
  4998.7 2071.51  4999.0 2073.16  5004.6 2073.16  5012.7 2078.81  5025.7 2082.21
  5036.2 2082.40  5041.6 2085.41  5057.1 2089.01  5065.0 2091.88  5070.5 2095.25
  5088.5 2097.70  5093.9 2099.90  5098.7 2100.05  5111.9 2098.66  5117.3 2099.96
  5123.8 2095.31  5134.7 2096.63  5140.8 2100.43  5169.6 2103.13  5179.2 2101.54
#Mann=5,-1,0
  4756.1    0.07       0  4994.2    0.07       0  4998.7    0.07       0
  5057.1    0.16       0  5098.7    0.07       0
Bank Sta=4994.2,4998.7
Exp/Cntr=0.3,0.1

Type RM Length L Ch R = 1,361,125,125,125
BEGIN DESCRIPTION:
Elm 76 4378
END DESCRIPTION:
XS GIS Cut Line= 3
      1531011.63      6764427.71      1531173.73      6764619.74
      1531295.42      6764712.97
#Sta/Elev= 30
  4748.7 2092.37  4793.8 2086.92  4808.1 2084.51  4822.4 2083.15  4828.9 2083.70
  4836.7 2081.99  4851.0 2080.54  4871.8 2079.87  4879.5 2080.41  4886.1 2078.64
  4893.0 2078.17  4900.4 2079.45  4906.9 2077.87  4914.7 2077.54  4929.0 2078.23
  4978.4 2077.64  4992.7 2076.01  4997.1 2073.19  5002.7 2073.19  5011.9 2071.28
  5012.2 2070.78  5016.4 2071.28  5021.2 2077.46  5027.4 2079.48  5035.7 2087.13
  5056.5 2097.70  5071.0 2098.71  5085.5 2101.24  5100.0 2102.20  5153.3 2102.84
#Mann=3,-1,0
  4748.7    0.07       0  5011.9    0.07       0  5016.4    0.07       0
Bank Sta=5011.9,5016.4
Exp/Cntr=0.3,0.1

Type RM Length L Ch R = 1,236,151,151,151
BEGIN DESCRIPTION:
Elm 76 4376
END DESCRIPTION:
XS GIS Cut Line= 3
      1530986.86      6764439.37      1531075.21      6764688.36
      1531204.29      6764762.99
#Sta/Elev= 30
  4735.8 2092.30  4778.6 2086.43  4840.5 2080.30  4896.8 2077.06  4904.1 2077.22
  4922.3 2072.83  4927.6 2073.28  4935.9 2072.07  4976.1 2070.90  4976.4 2070.40
  4980.6 2070.90  4984.1 2071.62  4989.4 2071.15  4997.2 2077.97  5007.4 2077.14
  5013.2 2084.19  5022.9 2085.12  5028.9 2083.27  5034.7 2087.72  5044.7 2086.71
  5066.2 2092.80  5072.0 2091.30  5087.8 2096.07  5093.6 2094.82  5103.6 2097.56
  5109.3 2096.00  5125.1 2098.44  5130.9 2096.97  5146.6 2099.29  5149.1 2098.90
#Mann=3,-1,0
  4735.8    0.07       0  4976.1    0.07       0  4980.6    0.07       0
Bank Sta=4976.1,4980.6
Exp/Cntr=0.3,0.1

Type RM Length L Ch R = 1,85,0,0,0
BEGIN DESCRIPTION:
Elm 76 4375
END DESCRIPTION:
XS GIS Cut Line= 3
      1530932.17      6764479.71      1530939.97      6764638.72
      1531065.00      6764763.01
#Sta/Elev= 30
  4840.8 2097.28  4879.1 2093.39  4909.2 2088.67  4949.2 2081.02  4959.2 2080.31
  4969.2 2075.22  4977.0 2069.50  4977.3 2069.00  4981.2 2069.00  4981.5 2069.50
  4997.1 2071.00  5017.2 2071.25  5031.3 2071.98  5038.4 2072.93  5045.5 2072.90
  5052.5 2073.75  5059.6 2073.25  5066.7 2074.57  5073.8 2074.08  5080.8 2075.31
  5087.9 2075.16  5095.0 2077.70  5102.1 2077.68  5109.1 2079.83  5137.4 2079.58
  5144.5 2080.08  5158.6 2079.80  5165.7 2079.16  5172.8 2079.88  5176.3 2079.34
#Mann=3,-1,0
  4840.8    0.07       0  4977.0    0.07       0  4981.5    0.07       0
Bank Sta=4977,4981.5
Exp/Cntr=0.3,0.1

Chan Stop Cuts=-1
