--- Elm 79.prj (project) ---

Proj Title=Elm 79 Base Level Engineering
Current Plan=p01
Default Exp/Contr=0.3,0.1
English Units
Geom File=g01
Flow File=f01
Plan File=p01
BEGIN DESCRIPTION:
Elm 79
END DESCRIPTION:

--- Elm 79.p01 (plan) ---

Plan Title=Multiple Run
Short Identifier=Multiple
Geom File=g01
Flow File=f01
Subcritical Flow
K Sum by GR= 0
Std Step Tol= 0.01
Critical Tol= 0.01
Num of Std Step Trials= 20
Max Error Tol= 0.3
Flow Tol Ratio= 0.001
Split Flow NTrial= 30
Split Flow Tol= 0.02
Split Flow Ratio= 0.02
Log Output Level= 0
Friction Slope Method= 1
Unsteady Friction Slope Method= 2
Unsteady Bridges Friction Slope Method= 1
Parabolic Critical Depth
Global Vel Dist=  1 , 1 , 1
Global Log Level= 0
CheckData=True
Encroach Param= -1, 0, 0, 0
BEGIN DESCRIPTION:
Multiple Run
END DESCRIPTION:

--- Elm 79.f01 (steady flow) ---

Flow Title=Multiple
Number of Profiles=7
Profile Names=10-year,25-year,50-year,1pct_min,100-year,1pct_plu,500-year
River Rch & RM= Elm 79,Reach-1,10863
     199     279     346     269     431     592     671
River Rch & RM= Elm 79,Reach-1,8834
     264     374     468     365     584     804     921
River Rch & RM= Elm 79,Reach-1,7268
     316     452     569     445     714     982    1140
River Rch & RM= Elm 79,Reach-1,5856
     385     555     703     552     885    1220    1420
River Rch & RM= Elm 79,Reach-1,2528
     405     585     741     582     933    1280    1500
River Rch & RM= Elm 79,Reach-1,553
     440     638     810     638    1020    1410    1650
Boundary for River Rch & Prof#=Elm 79,Reach-1,1
Up Type=0
Dn Type=3
Dn Slope=0.005
Boundary for River Rch & Prof#=Elm 79,Reach-1,2
Up Type=0
Dn Type=3
Dn Slope=0.005
Boundary for River Rch & Prof#=Elm 79,Reach-1,3
Up Type=0
Dn Type=3
Dn Slope=0.005
Boundary for River Rch & Prof#=Elm 79,Reach-1,4
Up Type=0
Dn Type=3
Dn Slope=0.005
Boundary for River Rch & Prof#=Elm 79,Reach-1,5
Up Type=0
Dn Type=3
Dn Slope=0.005
Boundary for River Rch & Prof#=Elm 79,Reach-1,6
Up Type=0
Dn Type=3
Dn Slope=0.005
Boundary for River Rch & Prof#=Elm 79,Reach-1,7
Up Type=0
Dn Type=3
Dn Slope=0.005

--- Elm 79.g01 (geometry) ---

Geom Title=Existing Conditions

River Reach=Elm 79,Reach-1
Reach XY= 30
      1537355.00      6762738.00      1537016.10      6763077.68
      1537035.63      6763258.09      1536540.88      6763501.39
      1536551.84      6763636.35      1536414.68      6763777.83
      1536255.09      6763695.28      1536061.97      6763784.67
      1536146.01      6763881.33      1536062.10      6763988.00
      1536197.23      6764134.59      1536112.50      6764288.00
      1536197.47      6764437.99      1535798.95      6765690.19
      1535405.00      6766038.00      1535551.93      6766146.30
      1535603.48      6766331.61      1535382.28      6766661.89
      1535015.47      6766928.18      1534949.17      6767190.30
      1534808.54      6767339.47      1534704.60      6767763.00
      1534757.07      6768132.14      1534854.40      6768248.62
      1534799.53      6768540.45      1534456.96      6768893.89
      1534449.53      6769240.45      1533856.23      6770098.51
      1533805.00      6770338.00      1534305.00      6770688.00

Type RM Length L Ch R = 1,10863,59,59,59
BEGIN DESCRIPTION:
Elm 79 4029
END DESCRIPTION:
XS GIS Cut Line= 3
      1537207.10      6762721.48      1537285.39      6762808.16
      1537373.78      6762877.75
#Sta/Elev= 30
  4883.2 2191.10  4900.6 2190.29  4907.3 2189.05  4914.8 2189.40  4921.5 2188.17
  4929.0 2188.05  4935.7 2186.87  4943.2 2186.13  4964.1 2185.13  4985.8 2182.11
  4992.5 2182.28  4996.5 2180.42  5002.9 2180.42  5006.8 2180.88  5013.2 2178.74
  5021.3 2174.00  5025.7 2172.63  5025.9 2172.13  5029.4 2172.13  5029.7 2172.63
  5035.7 2173.46  5042.1 2175.72  5050.2 2180.45  5056.6 2185.17  5063.1 2187.37
  5077.4 2190.24  5085.4 2190.64  5091.8 2192.04  5106.3 2194.22  5112.5 2194.44
#Mann=3,-1,0
  4883.2    0.16       0  5025.7    0.07       0  5029.7    0.16       0
Bank Sta=5025.7,5029.7
Exp/Cntr=0.3,0.1

Type RM Length L Ch R = 1,10804,91,91,91
BEGIN DESCRIPTION:
Elm 79 4028
END DESCRIPTION:
XS GIS Cut Line= 3
      1537155.01      6762773.56      1537243.74      6762850.14
      1537359.95      6762926.40
#Sta/Elev= 30
  4882.8 2194.55  4886.1 2194.55  4899.9 2192.45  4914.2 2189.44  4928.4 2187.11
  4935.6 2186.61  4942.7 2185.16  4949.3 2185.40  4956.9 2182.95  4963.6 2182.01
  4971.2 2177.40  4977.8 2174.20  4985.5 2174.36  4992.1 2171.71  5002.6 2171.25
  5004.4 2170.66  5004.6 2170.16  5008.1 2170.16  5008.4 2170.66  5013.5 2170.78
  5021.4 2171.81  5036.5 2174.66  5042.5 2178.79  5049.4 2182.56  5057.6 2185.71
  5063.6 2189.75  5072.7 2191.52  5108.9 2193.46  5114.9 2193.28  5139.0 2194.24
#Mann=3,-1,0
  4882.8    0.16       0  5004.4    0.07       0  5008.4    0.16       0
Bank Sta=5004.4,5008.4
Exp/Cntr=0.3,0.1

Type RM Length L Ch R = 1,10713,55,55,55
BEGIN DESCRIPTION:
Elm 79 4027
END DESCRIPTION:
XS GIS Cut Line= 3
      1537104.71      6762830.89      1537202.39      6762927.52
      1537320.88      6762985.00
#Sta/Elev= 30
  4862.6 2194.04  4867.8 2193.20  4874.9 2192.89  4882.0 2191.44  4903.2 2189.12
  4910.3 2188.76  4917.4 2187.43  4945.6 2184.04  4952.7 2179.90  4959.8 2168.91
  4971.9 2167.86  4972.2 2167.36  4975.7 2167.36  4975.9 2167.86  4981.0 2167.98
  4988.1 2172.22  4995.1 2170.76  4998.3 2174.03  5004.2 2174.03  5016.1 2179.37
  5038.6 2184.84  5047.4 2185.47  5055.7 2186.74  5061.2 2186.65  5078.2 2189.17
  5083.8 2189.03  5100.8 2190.64  5123.4 2192.07  5128.9 2191.80  5131.7 2192.61
#Mann=3,-1,0
  4862.6    0.16       0  4971.9    0.07       0  4975.9    0.16       0
Bank Sta=4971.9,4975.9
Exp/Cntr=0.3,0.1

Type RM Length L Ch R = 1,10658,84,84,84
BEGIN DESCRIPTION:
Elm 79 4026
END DESCRIPTION:
XS GIS Cut Line= 3
      1537057.85      6762877.78      1537172.08      6762971.58
      1537274.82      6763028.79
#Sta/Elev= 30
  4852.2 2193.17  4875.1 2191.64  4878.5 2191.17  4886.4 2191.07  4900.3 2189.77
  4913.7 2187.84  4921.6 2186.42  4942.4 2181.52  4950.3 2180.60  4956.7 2178.76
  4964.6 2178.27  4971.1 2174.80  4977.9 2173.77  4985.4 2170.03  4991.9 2168.13
  4996.7 2166.23  4996.9 2165.73  5000.4 2165.73  5000.7 2166.23  5006.0 2166.86
  5014.8 2172.87  5022.0 2179.75  5027.7 2180.86  5037.7 2183.56  5049.4 2184.61
  5059.7 2184.86  5065.4 2185.99  5087.2 2187.36  5094.9 2188.30  5117.6 2189.38
#Mann=4,-1,0
  4852.2    0.07       0  4875.1    0.16       0  4996.7    0.07       0
  5000.7    0.16       0
Bank Sta=4996.7,5000.7
Exp/Cntr=0.3,0.1

Type RM Length L Ch R = 1,10574,61,61,61
BEGIN DESCRIPTION:
Elm 79 4025
END DESCRIPTION:
XS GIS Cut Line= 3
      1537023.08      6762928.08      1537111.03      6763029.85
      1537212.64      6763093.87
#Sta/Elev= 30
  4865.5 2188.86  4874.0 2188.20  4880.6 2188.62  4888.3 2188.03  4909.2 2187.56
  4916.8 2187.02  4931.1 2184.49  4937.7 2181.56  4944.7 2179.22  4951.9 2178.65
  4958.5 2174.33  4966.2 2168.24  4972.8 2166.35  4978.4 2163.28  4978.7 2162.78
  4982.2 2162.78  4982.4 2163.28  4990.1 2163.63  5003.0 2164.10  5008.3 2173.00
  5023.6 2176.57  5029.5 2179.95  5044.7 2181.37  5060.0 2183.68  5065.9 2183.39
  5075.3 2184.81  5096.5 2186.62  5102.4 2185.94  5117.7 2185.82  5120.1 2185.01
#Mann=4,-1,0
  4865.5    0.07       0  4978.4    0.07       0  4982.4    0.07       0
  4990.1    0.16       0
Bank Sta=4978.4,4982.4
Exp/Cntr=0.3,0.1

Type RM Length L Ch R = 1,10513,49,49,49
BEGIN DESCRIPTION:
Elm 79 10513.132
END DESCRIPTION:
XS GIS Cut Line= 3
      1536971.00      6762969.76      1537052.17      6763043.86
      1537205.00      6763138.00
#Sta/Elev= 30
  4890.1 2184.21  4906.0 2183.56  4927.0 2178.53  4934.4 2181.26  4941.2 2179.08
  4948.6 2180.79  4955.3 2178.38  4962.8 2179.19  4969.5 2173.92  4976.8 2171.54
  4990.5 2162.55  4998.0 2161.49  4998.2 2160.99  5002.0 2161.49  5013.3 2163.92
  5026.8 2171.72  5034.6 2174.59  5050.0 2176.29  5055.9 2173.05  5071.3 2173.95
  5077.2 2171.87  5092.6 2178.33  5095.1 2177.64  5098.4 2176.72  5108.0 2179.49
  5113.8 2177.22  5129.2 2182.26  5135.1 2181.28  5150.5 2183.10  5179.5 2182.00
#Mann=4,-1,0
  4890.1    0.07       0  4998.0    0.07       0  5002.0    0.07       0
  5095.1    0.16       0
Bank Sta=4998,5002
Exp/Cntr=0.3,0.1

Type RM Length L Ch R = 1,10464,73,73,73
BEGIN DESCRIPTION:
Elm 79 10464.12
END DESCRIPTION:
XS GIS Cut Line= 3
      1536931.06      6763023.58      1537019.63      6763079.15
      1537189.75      6763148.58
#Sta/Elev= 30
  4899.1 2183.45  4904.4 2183.45  4913.2 2178.77  4919.1 2177.98  4934.5 2172.01
  4940.4 2171.11  4955.7 2167.05  4971.0 2161.40  4976.9 2160.53  5018.3 2160.31
  5018.5 2159.81  5022.3 2160.31  5031.1 2164.37  5038.4 2166.51  5043.8 2163.00
  5062.4 2163.51  5067.8 2161.70  5085.1 2162.38  5091.9 2163.66  5097.3 2162.67
  5106.7 2165.12  5115.9 2168.82  5121.3 2168.04  5128.3 2172.22  5145.3 2177.98
  5146.5 2177.82  5150.7 2177.24  5169.3 2180.47  5174.7 2179.05  5187.4 2180.20
#Mann=4,-1,0
  4899.1    0.07       0  5018.3    0.07       0  5022.3    0.07       0
  5146.5    0.16       0
Bank Sta=5018.3,5022.3
Exp/Cntr=0.3,0.1

Type RM Length L Ch R = 1,10391,60,60,60
BEGIN DESCRIPTION:
Elm 79 10390.96
END DESCRIPTION:
XS GIS Cut Line= 3
      1536901.54      6763084.35      1537047.41      6763138.18
      1537189.77      6763155.54
#Sta/Elev= 30
  4845.0 2182.73  4849.5 2182.73  4867.3 2180.97  4872.7 2180.85  4891.3 2176.80
  4897.8 2174.62  4903.1 2175.37  4912.6 2172.51  4922.9 2170.12  4928.2 2170.75
  4934.0 2167.92  4951.3 2163.90  4951.5 2163.40  4955.0 2163.40  4955.3 2163.90
  4958.6 2166.72  4976.6 2164.36  4983.7 2163.92  4989.1 2167.28  5018.2 2166.32
  5028.3 2165.36  5036.8 2165.10  5041.8 2168.59  5068.6 2168.72  5078.6 2170.28
  5114.8 2177.44  5118.4 2178.21  5123.4 2176.86  5129.0 2178.41  5143.9 2179.00
#Mann=4,-1,0
  4845.0    0.07       0  4951.3    0.07       0  4955.3    0.07       0
  5114.8    0.16       0
Bank Sta=4951.3,4955.3
Exp/Cntr=0.3,0.1

Type RM Length L Ch R = 1,10331,63,63,63
BEGIN DESCRIPTION:
Elm 79 10331.08
END DESCRIPTION:
XS GIS Cut Line= 3
      1536908.56      6763148.61      1537010.95      6763186.79
      1537180.59      6763191.98
#Sta/Elev= 30
  4888.1 2179.29  4895.0 2179.02  4916.3 2176.21  4930.8 2175.33  4937.7 2174.31
  4948.3 2173.90  4955.8 2174.40  4961.1 2173.34  4980.4 2173.71  4986.1 2174.67
  4991.4 2172.80  4996.9 2173.63  5001.9 2173.63  5009.4 2171.52  5009.7 2171.02
  5013.2 2171.02  5013.4 2171.52  5021.4 2172.41  5031.4 2175.06  5051.5 2176.46
  5061.5 2176.57  5071.5 2177.04  5081.5 2176.93  5111.5 2177.55  5131.5 2177.49
  5141.5 2176.49  5151.5 2176.43  5161.5 2177.73  5166.4 2178.67  5167.1 2178.80
#Mann=4,-1,0
  4888.1    0.07       0  5009.4    0.07       0  5013.4    0.07       0
  5166.4    0.16       0
Bank Sta=5009.4,5013.4
Exp/Cntr=0.3,0.1

Type RM Length L Ch R = 1,10268,57,57,57
BEGIN DESCRIPTION:
Elm 79 10267.62
END DESCRIPTION:
XS GIS Cut Line= 3
      1536955.43      6763198.96      1537045.67      6763238.87
      1537165.50      6763224.98
#Sta/Elev= 30
  4900.6 2172.39  4903.1 2172.39  4913.6 2169.47  4922.0 2170.17  4931.4 2170.18
  4936.9 2169.33  4943.9 2171.57  4954.7 2170.73  4960.1 2167.40  4965.7 2162.44
  4976.7 2157.55  4983.4 2154.13  4986.9 2151.81  4987.2 2151.31  4990.7 2151.31
  4990.9 2151.81  4996.2 2152.08  5001.5 2152.08  5008.7 2153.04  5018.7 2153.74
  5028.8 2154.17  5038.9 2161.37  5047.1 2167.90  5052.1 2171.41  5059.0 2171.62
  5069.1 2171.11  5079.1 2170.95  5089.2 2171.44  5117.1 2173.83  5119.9 2173.83
#Mann=3,-1,0
  4900.6    0.07       0  4986.9    0.07       0  4990.9    0.07       0
Bank Sta=4986.9,4990.9
Exp/Cntr=0.3,0.1

Type RM Length L Ch R = 1,10211,77,77,77
BEGIN DESCRIPTION:
Elm 79 10210.71
END DESCRIPTION:
XS GIS Cut Line= 3
      1536950.20      6763205.91      1537009.22      6763280.54
      1537118.58      6763365.60
#Sta/Elev= 30
  4902.0 2171.53  4914.4 2170.87  4928.9 2167.91  4942.9 2167.99  4949.7 2165.70
  4956.0 2166.55  4964.1 2163.48  4968.8 2159.68  4978.5 2153.49  4984.9 2151.38
  4990.3 2151.21  4990.6 2150.71  4994.1 2150.71  4994.3 2151.21  4997.1 2151.21
  4999.6 2153.68  5006.0 2154.01  5014.1 2156.26  5020.5 2156.49  5028.6 2159.46
  5038.3 2161.64  5049.4 2165.98  5055.8 2167.24  5063.9 2170.24  5070.2 2170.56
  5092.9 2176.06  5113.7 2181.93  5120.0 2181.65  5128.1 2182.63  5135.7 2182.09
#Mann=5,-1,0
  4902.0    0.07       0  4968.8    0.16       0  4990.3    0.07       0
  4994.3    0.16       0  5038.3    0.07       0
Bank Sta=4990.3,4994.3
Exp/Cntr=0.3,0.1

Type RM Length L Ch R = 1,10134,114,114,114
BEGIN DESCRIPTION:
Elm 79 10134.38
END DESCRIPTION:
XS GIS Cut Line= 3
      1536938.03      6763211.05      1536955.40      6763339.57
      1536945.10      6763444.28
#Sta/Elev= 30
  4881.0 2175.19  4888.0 2173.92  4894.4 2173.30  4899.4 2171.60  4908.2 2170.34
  4918.3 2168.38  4928.4 2165.46  4934.2 2163.55  4948.6 2158.94  4958.6 2156.27
  4967.0 2153.56  4972.1 2153.62  4978.8 2151.08  4986.9 2150.18  4987.2 2149.68
  4990.7 2149.68  4990.9 2150.18  4999.0 2150.27  5007.4 2151.64  5010.7 2151.64
  5019.2 2156.81  5029.2 2159.27  5039.8 2164.53  5059.4 2170.55  5065.1 2172.89
  5070.1 2172.91  5079.4 2174.64  5089.5 2175.55  5109.6 2176.13  5115.9 2175.94
#Mann=5,-1,0
  4881.0    0.07       0  4934.2    0.16       0  4986.9    0.07       0
  4990.9    0.16       0  5039.8    0.07       0
Bank Sta=4986.9,4990.9
Exp/Cntr=0.3,0.1

Type RM Length L Ch R = 1,10020,102,102,102
BEGIN DESCRIPTION:
Elm 79 10020.38
END DESCRIPTION:
XS GIS Cut Line= 3
      1536839.08      6763212.86      1536854.70      6763296.17
      1536925.88      6763429.84
#Sta/Elev= 30
  4918.8 2178.54  4926.4 2178.94  4934.2 2177.94  4944.4 2174.39  4954.5 2169.34
  4964.7 2163.83  4973.9 2157.55  4979.0 2158.50  4982.0 2155.78  4985.1 2152.96
  4995.2 2147.17  4999.9 2145.22  5000.2 2144.72  5003.7 2144.72  5003.9 2145.22
  5007.4 2145.22  5013.1 2147.80  5018.7 2148.53  5028.3 2150.33  5050.9 2157.24
  5062.7 2161.66  5073.3 2161.76  5079.0 2162.90  5100.9 2165.44  5107.6 2167.01
  5117.2 2168.65  5119.9 2169.51  5130.3 2172.19  5144.9 2174.23  5155.0 2174.56
#Mann=5,-1,0
  4918.8    0.07       0  4982.0    0.16       0  4999.9    0.07       0
  5003.9    0.16       0  5119.9    0.07       0
Bank Sta=4999.9,5003.9
Exp/Cntr=0.3,0.1

Type RM Length L Ch R = 1,9918,52,52,52
BEGIN DESCRIPTION:
Elm 79 9918.19
END DESCRIPTION:
XS GIS Cut Line= 3
      1536759.21      6763264.90      1536806.09      6763384.71
      1536872.03      6763445.44
#Sta/Elev= 30
  4881.5 2174.32  4886.9 2176.24  4903.0 2172.12  4906.0 2171.23  4911.4 2171.62
  4917.0 2168.47  4935.9 2162.31  4941.2 2162.47  4949.3 2159.16  4960.0 2155.77
  4965.7 2152.66  4971.0 2150.97  4990.1 2147.55  4995.5 2143.63  5001.0 2142.63
  5001.2 2142.13  5004.7 2142.13  5005.0 2142.63  5012.8 2142.84  5018.9 2147.83
  5025.7 2150.96  5033.1 2155.09  5054.1 2163.11  5061.5 2165.09  5068.3 2167.69
  5075.6 2168.13  5082.8 2170.55  5089.8 2170.74  5096.6 2171.70  5099.8 2171.56
#Mann=5,-1,0
  4881.5    0.07       0  4903.0    0.16       0  5001.0    0.07       0
  5005.0    0.16       0  5082.8    0.07       0
Bank Sta=5001,5005
Exp/Cntr=0.3,0.1

Type RM Length L Ch R = 1,9866,70,70,70
BEGIN DESCRIPTION:
Elm 79 9865.89
END DESCRIPTION:
XS GIS Cut Line= 3
      1536689.79      6763303.14      1536755.74      6763391.65
      1536814.75      6763499.25
#Sta/Elev= 30
  4888.1 2170.38  4894.4 2168.00  4917.4 2162.18  4938.2 2159.51  4944.5 2159.38
  4952.8 2157.28  4959.1 2154.93  4973.7 2148.27  4988.3 2146.12  4993.7 2147.28
  5003.7 2147.34  5009.4 2146.69  5017.1 2142.17  5023.5 2140.49  5023.7 2139.99
  5027.2 2139.99  5027.5 2140.49  5039.9 2148.62  5047.3 2154.15  5053.0 2156.90
  5062.7 2162.86  5069.1 2167.39  5074.8 2169.36  5085.2 2171.76  5090.9 2171.63
  5093.3 2172.11  5097.0 2172.85  5107.0 2173.02  5112.7 2172.76  5121.2 2173.10
#Mann=4,-1,0
  4888.1    0.16       0  5023.5    0.07       0  5027.5    0.16       0
  5093.3    0.07       0
Bank Sta=5023.5,5027.5
Exp/Cntr=0.3,0.1

Type RM Length L Ch R = 1,9796,65,65,65
BEGIN DESCRIPTION:
Elm 79 9795.63
END DESCRIPTION:
XS GIS Cut Line= 3
      1536630.72      6763346.48      1536701.92      6763436.79
      1536769.82      6763513.17
#Sta/Elev= 30
  4881.7 2175.90  4885.9 2175.90  4893.3 2172.54  4899.7 2171.16  4907.8 2165.98
  4914.2 2164.52  4921.8 2160.28  4928.6 2157.09  4935.0 2157.21  4943.0 2156.54
  4957.5 2156.13  4971.9 2150.22  4978.3 2142.20  4990.7 2137.92  4991.0 2137.42
  4994.5 2137.42  4994.7 2137.92  4995.2 2142.17  5000.9 2142.17  5006.9 2145.75
  5013.6 2150.21  5021.2 2153.07  5027.8 2156.20  5042.1 2159.94  5049.6 2163.36
  5056.3 2165.44  5063.8 2168.71  5078.0 2171.01  5085.6 2171.82  5098.9 2173.10
#Mann=4,-1,0
  4881.7    0.16       0  4990.7    0.07       0  4994.7    0.16       0
  5085.6    0.07       0
Bank Sta=4990.7,4994.7
Exp/Cntr=0.3,0.1

Type RM Length L Ch R = 1,9731,104,104,104
BEGIN DESCRIPTION:
Elm 79 9730.57
END DESCRIPTION:
XS GIS Cut Line= 3
      1536566.54      6763374.32      1536658.52      6763485.40
      1536736.67      6763547.92
#Sta/Elev= 30
  4860.2 2173.00  4868.5 2173.44  4876.4 2170.25  4882.9 2169.04  4890.7 2164.74
  4897.2 2163.20  4903.9 2159.12  4911.5 2155.92  4940.2 2153.83  4946.7 2154.92
  4954.5 2152.06  4961.0 2152.86  4968.8 2150.56  4975.4 2147.08  4981.9 2149.06
  4989.7 2143.83  4996.2 2143.18  5002.9 2138.44  5009.5 2137.22  5009.7 2136.72
  5013.5 2137.22  5025.5 2142.12  5038.7 2150.68  5046.7 2153.20  5061.1 2161.11
  5075.5 2165.97  5081.0 2166.18  5096.3 2170.17  5100.5 2168.88  5104.5 2168.88
#Mann=4,-1,0
  4860.2    0.16       0  5009.5    0.07       0  5013.5    0.16       0
  5081.0    0.07       0
Bank Sta=5009.5,5013.5
Exp/Cntr=0.3,0.1

Type RM Length L Ch R = 1,9627,61,61,61
BEGIN DESCRIPTION:
Elm 79 9626.89
END DESCRIPTION:
XS GIS Cut Line= 3
      1536510.96      6763402.09      1536563.04      6763513.18
      1536706.93      6763553.05
#Sta/Elev= 30
  4899.6 2169.04  4906.1 2166.37  4921.8 2162.52  4928.2 2158.14  4939.1 2154.42
  4944.6 2153.13  4950.3 2149.30  4961.3 2146.18  4967.4 2142.42  4973.0 2140.45
  4983.4 2135.59  4988.3 2135.19  4988.5 2134.69  4992.0 2134.69  4992.3 2135.19
  5005.5 2143.88  5013.5 2148.36  5018.6 2148.37  5022.2 2152.33  5032.2 2152.56
  5059.9 2152.82  5065.8 2154.48  5086.6 2158.32  5094.1 2158.38  5099.3 2157.58
  5128.1 2158.14  5148.8 2159.50  5159.0 2160.95  5167.9 2162.90  5171.6 2161.93
#Mann=6,-1,0
  4899.6    0.16       0  4988.3    0.07       0  4992.3    0.16       0
  5013.5    0.07       0  5032.2    0.16       0  5159.0    0.07       0
Bank Sta=4988.3,4992.3
Exp/Cntr=0.3,0.1

Type RM Length L Ch R = 1,9566,75,75,75
BEGIN DESCRIPTION:
Elm 79 9565.9
END DESCRIPTION:
XS GIS Cut Line= 3
      1536332.17      6763492.35      1536516.16      6763537.48
      1536721.39      6763559.90
#Sta/Elev= 30
  4814.1 2166.77  4819.5 2166.75  4847.9 2158.08  4855.9 2154.71  4861.1 2154.30
  4868.5 2151.75  4920.0 2150.99  4939.1 2153.96  4944.2 2153.33  4961.2 2155.87
  4971.5 2155.93  4980.7 2151.65  4985.8 2151.36  4992.1 2143.88  4998.4 2134.63
  4998.6 2134.13  5002.4 2134.63  5011.4 2136.96  5022.5 2145.68  5032.6 2149.84
  5042.6 2152.16  5067.6 2151.97  5082.9 2152.02  5113.0 2155.63  5142.3 2157.30
  5147.3 2156.38  5163.3 2157.09  5174.2 2159.03  5193.5 2161.93  5210.0 2165.88
#Mann=6,-1,0
  4814.1    0.16       0  4998.4    0.07       0  5002.4    0.16       0
  5011.4    0.07       0  5067.6    0.16       0  5174.2    0.07       0
Bank Sta=4998.4,5002.4
Exp/Cntr=0.3,0.1

Type RM Length L Ch R = 1,9491,64,64,64
BEGIN DESCRIPTION:
Elm 79 9490.99
END DESCRIPTION:
XS GIS Cut Line= 3
      1536373.84      6763537.50      1536545.67      6763598.25
      1536736.63      6763586.10
#Sta/Elev= 30
  4810.6 2151.31  4833.0 2147.94  4889.2 2149.63  4914.9 2153.11  4926.9 2153.22
  4939.1 2153.96  4945.8 2151.01  4951.1 2151.86  4960.3 2147.54  4970.9 2139.16
  4976.7 2132.78  4982.0 2134.75  4987.8 2132.49  4988.1 2131.99  4991.8 2132.49
  4995.0 2132.49  5002.2 2136.96  5012.2 2139.94  5022.2 2140.79  5040.0 2135.79
  5042.3 2134.95  5052.3 2137.83  5062.3 2138.24  5071.4 2136.67  5076.4 2141.55
  5081.1 2143.85  5112.4 2147.25  5142.5 2155.72  5172.5 2169.28  5184.2 2170.64
#Mann=6,-1,0
  4810.6    0.16       0  4926.9    0.07       0  4987.8    0.07       0
  4991.8    0.07       0  5040.0    0.16       0  5081.1    0.07       0
Bank Sta=4987.8,4991.8
Exp/Cntr=0.3,0.1

Type RM Length L Ch R = 1,9427,85,85,85
BEGIN DESCRIPTION:
Elm 79 9426.97
END DESCRIPTION:
XS GIS Cut Line= 3
      1536398.07      6763553.08      1536540.47      6763659.01
      1536625.52      6763719.77
#Sta/Elev= 30
  4827.0 2147.56  4842.7 2148.96  4849.0 2148.43  4857.4 2149.09  4878.2 2148.78
  4885.5 2149.29  4892.8 2151.00  4899.0 2150.77  4922.0 2152.01  4949.1 2148.34
  4978.3 2147.92  4999.1 2135.30  5002.2 2132.09  5002.4 2131.59  5005.9 2131.59
  5006.2 2132.09  5022.3 2133.07  5028.5 2137.79  5034.7 2139.19  5043.3 2146.29
  5049.4 2148.40  5058.0 2155.84  5064.1 2157.76  5072.8 2162.77  5078.9 2165.05
  5085.0 2164.32  5093.6 2166.03  5099.8 2164.49  5105.6 2166.22  5109.0 2166.22
#Mann=4,-1,0
  4827.0    0.16       0  5002.2    0.07       0  5006.2    0.16       0
  5072.8    0.07       0
Bank Sta=5002.2,5006.2
Exp/Cntr=0.3,0.1

Type RM Length L Ch R = 1,9342,96,96,96
BEGIN DESCRIPTION:
Elm 79 9341.59
END DESCRIPTION:
XS GIS Cut Line= 3
      1536410.25      6763589.55      1536476.23      6763716.30
      1536538.05      6763803.88
#Sta/Elev= 30
  4856.7 2146.25  4866.2 2145.74  4874.8 2146.56  4880.5 2147.88  4888.8 2148.85
  4902.6 2149.91  4919.0 2151.69  4924.7 2151.16  4946.8 2146.39  4968.9 2145.96
  4979.0 2144.88  4985.4 2141.82  4994.9 2131.41  4995.7 2130.51  4996.0 2130.01
  4999.5 2130.01  4999.7 2130.51  5007.0 2130.94  5013.9 2130.75  5021.8 2133.59
  5027.9 2138.41  5036.5 2144.66  5042.7 2149.86  5050.6 2155.25  5063.6 2163.57
  5072.2 2162.82  5078.4 2164.82  5087.0 2164.91  5093.2 2165.96  5106.8 2166.13
#Mann=4,-1,0
  4856.7    0.16       0  4994.9    0.07       0  4995.7    0.07       0
  4999.7    0.07       0
Bank Sta=4995.7,4999.7
Exp/Cntr=0.3,0.1

Type RM Length L Ch R = 1,9246,75,75,75
BEGIN DESCRIPTION:
Elm 79 9246.27
END DESCRIPTION:
XS GIS Cut Line= 3
      1536405.05      6763634.75      1536406.79      6763780.54
      1536449.80      6763873.46
#Sta/Elev= 30
  4852.3 2150.42  4856.4 2150.42  4865.6 2151.67  4875.6 2151.53  4885.6 2150.23
  4905.6 2147.05  4915.6 2143.55  4925.6 2139.47  4927.8 2139.14  4935.6 2137.95
  4955.6 2133.20  4965.6 2132.81  4975.6 2130.93  4985.6 2129.41  4992.3 2129.01
  4992.6 2128.51  4996.1 2128.51  4996.3 2129.01  4998.1 2129.01  5008.8 2135.12
  5017.3 2145.82  5026.2 2154.49  5031.7 2155.95  5039.4 2162.00  5049.1 2162.78
  5054.6 2163.40  5072.0 2163.50  5077.6 2164.05  5083.5 2164.02  5100.5 2164.63
#Mann=4,-1,0
  4852.3    0.16       0  4927.8    0.07       0  4992.3    0.07       0
  4996.3    0.07       0
Bank Sta=4992.3,4996.3
Exp/Cntr=0.3,0.1

Type RM Length L Ch R = 1,9171,110,110,110
BEGIN DESCRIPTION:
Elm 79 9170.76
END DESCRIPTION:
XS GIS Cut Line= 3
      1536318.25      6763605.21      1536339.08      6763778.80
      1536380.38      6763861.41
#Sta/Elev= 30
  4832.9 2148.44  4844.2 2147.31  4855.9 2144.65  4876.0 2136.97  4886.1 2134.60
  4896.1 2133.47  4906.2 2133.38  4916.3 2134.82  4926.4 2137.20  4931.5 2134.91
  4936.6 2134.96  4946.5 2131.10  4956.6 2128.73  4976.7 2129.35  4996.9 2128.62
  5004.8 2130.96  5007.7 2130.96  5009.1 2128.47  5009.4 2127.97  5012.9 2127.97
  5013.1 2128.47  5027.9 2137.95  5033.5 2137.29  5040.4 2147.14  5050.2 2153.74
  5062.7 2157.58  5072.6 2157.01  5078.2 2159.06  5095.0 2159.10  5100.1 2160.14
#Mann=4,-1,0
  4832.9    0.16       0  4936.6    0.07       0  5009.1    0.07       0
  5013.1    0.07       0
Bank Sta=5009.1,5013.1
Exp/Cntr=0.3,0.1

Type RM Length L Ch R = 1,9061,78,78,78
BEGIN DESCRIPTION:
Elm 79 9061.33
END DESCRIPTION:
XS GIS Cut Line= 3
      1536255.74      6763600.00      1536259.22      6763728.46
      1536344.29      6763856.94
#Sta/Elev= 30
  4902.9 2153.45  4915.9 2149.78  4960.9 2139.44  4970.9 2138.25  4980.9 2134.99
  4990.9 2129.57  5000.9 2129.23  5009.2 2131.31  5020.9 2133.18  5034.8 2134.47
  5042.9 2132.02  5049.9 2126.23  5068.9 2125.76  5069.2 2125.26  5072.7 2125.26
  5072.9 2125.76  5078.8 2127.65  5086.0 2132.51  5092.0 2132.98  5101.0 2137.65
  5107.0 2136.52  5122.1 2148.35  5128.1 2143.13  5137.2 2146.03  5143.1 2143.06
  5150.8 2151.62  5158.2 2155.94  5164.2 2155.41  5173.3 2156.22  5185.5 2156.17
#Mann=5,-1,0
  4902.9    0.07       0  4915.9    0.16       0  5009.2    0.07       0
  5068.9    0.07       0  5072.9    0.07       0
Bank Sta=5068.9,5072.9
Exp/Cntr=0.3,0.1

Type RM Length L Ch R = 1,8983,149,149,149
BEGIN DESCRIPTION:
Elm 79 8983.32
END DESCRIPTION:
XS GIS Cut Line= 3
      1536182.83      6763606.94      1536194.98      6763740.61
      1536298.59      6763823.50
#Sta/Elev= 30
  4870.2 2149.65  4873.2 2149.65  4881.3 2147.98  4891.3 2145.24  4921.5 2138.72
  4941.5 2132.23  4948.0 2130.89  4953.0 2132.43  4968.0 2126.38  4971.7 2124.94
  4998.6 2124.05  4998.8 2123.55  5002.3 2123.55  5002.6 2124.05  5003.2 2124.05
  5009.5 2125.00  5017.2 2124.33  5024.0 2125.39  5038.4 2124.39  5044.8 2125.38
  5052.8 2125.18  5059.2 2133.19  5067.2 2132.45  5073.6 2139.19  5088.0 2139.68
  5094.4 2143.75  5102.4 2145.28  5108.8 2145.61  5123.2 2148.76  5137.1 2149.77
#Mann=5,-1,0
  4870.2    0.07       0  4968.0    0.16       0  4998.6    0.07       0
  5002.6    0.16       0  5003.2    0.07       0
Bank Sta=4998.6,5002.6
Exp/Cntr=0.3,0.1

Type RM Length L Ch R = 1,8834,95,95,95
BEGIN DESCRIPTION:
Elm 79 8834.19
END DESCRIPTION:
XS GIS Cut Line= 3
      1535891.15      6763737.14      1536063.04      6763780.54
      1536306.10      6763830.89
#Sta/Elev= 30
  4821.6 2155.99  4826.2 2155.99  4843.3 2152.30  4848.5 2153.71  4856.5 2149.06
  4884.3 2141.34  4908.1 2141.11  4925.4 2136.58  4930.6 2137.01  4966.4 2130.91
  4971.6 2132.89  4990.6 2132.44  4997.3 2133.29  5008.5 2132.75  5035.3 2133.80
  5058.7 2133.55  5063.8 2129.23  5080.6 2128.90  5080.8 2128.40  5084.6 2128.90
  5108.9 2133.33  5114.0 2129.77  5123.5 2131.95  5153.9 2135.75  5164.3 2138.48
  5174.5 2138.97  5194.9 2141.93  5209.2 2144.23  5225.6 2148.79  5247.1 2151.22
#Mann=5,-1,0
  4821.6   0.035       0  5035.3    0.16       0  5080.6   0.035       0
  5084.6    0.16       0  5123.5    0.07       0
Bank Sta=5080.6,5084.6
Exp/Cntr=0.3,0.1

Type RM Length L Ch R = 1,8739,120,120,120
BEGIN DESCRIPTION:
Elm 79 8739.43
END DESCRIPTION:
XS GIS Cut Line= 3
      1535953.65      6763881.24      1536122.06      6763851.72
      1536310.64      6763886.32
#Sta/Elev= 30
  4831.8 2145.47  4863.6 2143.63  4873.8 2142.35  4884.3 2140.49  4904.2 2134.74
  4929.3 2132.61  4938.6 2132.21  4944.8 2130.42  4955.0 2125.61  4965.1 2122.52
  4977.1 2121.12  4996.0 2120.62  4996.3 2120.12  4999.8 2120.12  5000.0 2120.62
  5015.9 2120.63  5026.1 2121.30  5036.3 2123.49  5058.3 2126.65  5063.5 2128.21
  5068.6 2128.46  5097.3 2134.76  5107.4 2137.08  5116.6 2139.79  5121.7 2138.21
  5127.8 2140.81  5168.4 2150.26  5174.8 2151.25  5179.9 2150.15  5194.5 2153.62
#Mann=6,-1,0
  4831.8    0.07       0  4929.3   0.035       0  4977.1    0.16       0
  4996.0    0.07       0  5000.0    0.16       0  5058.3    0.07       0
Bank Sta=4996,5000
Exp/Cntr=0.3,0.1

Type RM Length L Ch R = 1,8619,116,116,116
BEGIN DESCRIPTION:
Elm 79 8618.95
END DESCRIPTION:
XS GIS Cut Line= 3
      1535946.76      6763903.82      1536101.23      6763943.73
      1536328.66      6763940.26
#Sta/Elev= 30
  4842.0 2144.95  4871.2 2143.55  4877.5 2142.44  4902.2 2140.07  4912.5 2138.41
  4918.2 2136.22  4923.3 2136.21  4933.1 2134.16  4953.6 2129.09  4958.8 2129.87
  4964.1 2127.23  4974.5 2125.45  4984.8 2124.93  4994.3 2123.70  5016.0 2122.98
  5035.3 2122.48  5045.0 2121.62  5048.0 2120.42  5048.3 2119.92  5051.8 2119.92
  5052.0 2120.42  5065.0 2120.55  5085.3 2120.98  5125.3 2128.74  5135.3 2129.38
  5165.3 2138.44  5195.3 2145.97  5215.3 2150.73  5224.7 2152.23  5229.0 2152.23
#Mann=5,-1,0
  4842.0    0.07       0  5016.0    0.16       0  5048.0    0.07       0
  5052.0    0.16       0  5065.0    0.07       0
Bank Sta=5048,5052
Exp/Cntr=0.3,0.1

Type RM Length L Ch R = 1,8503,80,80,80
BEGIN DESCRIPTION:
Elm 79 8502.89
END DESCRIPTION:
XS GIS Cut Line= 3
      1535997.02      6764018.38      1536102.97      6764032.28
      1536328.65      6764037.48
#Sta/Elev= 30
  4897.9 2138.06  4926.1 2135.93  4932.3 2134.37  4937.3 2135.24  4956.4 2130.85
  4966.5 2129.48  4976.6 2129.97  4986.6 2131.81  4996.7 2129.90  5003.3 2127.23
  5008.3 2127.23  5016.8 2124.94  5026.8 2123.91  5034.0 2120.34  5039.0 2121.85
  5056.8 2117.14  5064.8 2116.19  5065.1 2115.69  5068.6 2115.69  5068.8 2116.19
  5096.8 2117.38  5106.8 2119.08  5116.8 2123.66  5126.8 2126.12  5146.8 2134.06
  5166.8 2146.72  5176.8 2152.32  5196.8 2151.22  5226.2 2154.90  5230.5 2154.90
#Mann=3,-1,0
  4897.9    0.07       0  5064.8    0.07       0  5068.8    0.07       0
Bank Sta=5064.8,5068.8
Exp/Cntr=0.3,0.1

Type RM Length L Ch R = 1,8423,74,74,74
BEGIN DESCRIPTION:
Elm 79 8422.83
END DESCRIPTION:
XS GIS Cut Line= 3
      1535990.12      6764086.10      1536155.05      6764087.83
      1536325.23      6764082.62
#Sta/Elev= 30
  4834.8 2139.20  4839.7 2139.20  4849.7 2138.37  4859.7 2137.27  4879.7 2135.53
  4899.7 2133.52  4909.7 2133.17  4929.7 2130.55  4939.7 2128.72  4949.7 2127.27
  4959.7 2123.32  4969.7 2117.90  4979.7 2116.77  4989.7 2117.71  4997.2 2114.51
  5019.7 2114.61  5027.7 2114.21  5028.0 2113.71  5031.5 2113.71  5031.7 2114.21
  5059.7 2114.50  5069.7 2116.24  5079.7 2120.78  5099.7 2131.90  5129.8 2148.19
  5139.8 2153.82  5156.2 2162.28  5161.2 2160.72  5167.4 2162.23  5170.0 2162.23
#Mann=3,-1,0
  4834.8    0.07       0  5027.7    0.07       0  5031.7    0.07       0
Bank Sta=5027.7,5031.7
Exp/Cntr=0.3,0.1

Type RM Length L Ch R = 1,8349,61,61,61
BEGIN DESCRIPTION:
Elm 79 8349.12
END DESCRIPTION:
XS GIS Cut Line= 3
      1535997.08      6764136.44      1536198.45      6764145.12
      1536321.69      6764136.56
#Sta/Elev= 30
  4802.4 2138.55  4850.4 2132.91  4860.4 2132.11  4870.4 2131.99  4880.4 2130.97
  4890.4 2128.40  4900.4 2126.95  4910.4 2123.46  4919.7 2119.40  4930.4 2117.99
  4940.4 2117.31  4950.1 2117.36  4955.1 2114.33  4960.5 2113.40  4997.7 2111.83
  4998.0 2111.33  5001.5 2111.33  5001.7 2111.83  5010.5 2111.88  5020.5 2114.28
  5030.1 2117.96  5035.1 2116.77  5040.6 2121.26  5080.7 2141.32  5090.7 2147.43
  5100.7 2154.00  5110.8 2159.34  5115.9 2161.26  5120.8 2163.11  5127.5 2163.72
#Mann=5,-1,0
  4802.4    0.07       0  4919.7    0.16       0  4997.7    0.07       0
  5001.7    0.16       0  5115.9    0.07       0
Bank Sta=4997.7,5001.7
Exp/Cntr=0.3,0.1

Type RM Length L Ch R = 1,8288,111,111,111
BEGIN DESCRIPTION:
Elm 79 8287.85
END DESCRIPTION:
XS GIS Cut Line= 3
      1535983.14      6764204.15      1536158.52      6764193.73
      1536301.34      6764226.43
#Sta/Elev= 30
  4824.3 2138.34  4827.8 2138.34  4836.2 2137.60  4842.5 2136.66  4847.5 2136.79
  4866.2 2134.03  4886.3 2132.12  4906.3 2131.09  4926.3 2127.81  4936.4 2125.02
  4956.4 2115.93  4963.2 2113.19  4966.4 2111.90  5004.6 2110.43  5004.9 2109.93
  5008.4 2109.93  5008.6 2110.43  5016.9 2110.52  5036.9 2117.25  5042.0 2119.24
  5047.7 2122.68  5078.4 2133.65  5084.9 2139.03  5090.1 2139.62  5099.0 2144.52
  5109.2 2148.92  5119.5 2152.87  5127.9 2156.71  5140.0 2161.14  5146.5 2161.22
#Mann=4,-1,0
  4824.3    0.07       0  4963.2    0.16       0  5004.6    0.07       0
  5008.6    0.16       0
Bank Sta=5004.6,5008.6
Exp/Cntr=0.3,0.1

Type RM Length L Ch R = 1,8177,86,86,86
BEGIN DESCRIPTION:
Elm 79 8176.79
END DESCRIPTION:
XS GIS Cut Line= 3
      1535969.24      6764266.64      1536113.38      6764290.96
      1536297.44      6764275.33
#Sta/Elev= 30
  4853.3 2138.41  4869.3 2136.91  4893.1 2135.34  4899.7 2133.98  4909.8 2132.75
  4930.1 2131.33  4940.3 2131.43  4948.5 2129.74  4953.6 2129.66  4980.8 2111.61
  4989.0 2109.69  4989.2 2109.19  4992.7 2109.19  4993.0 2109.69  5020.7 2110.15
  5031.2 2109.85  5041.2 2110.35  5061.3 2115.97  5071.4 2118.43  5081.4 2121.67
  5090.0 2125.56  5095.0 2125.90  5101.5 2130.66  5121.5 2139.51  5131.6 2144.73
  5141.6 2150.41  5151.6 2155.26  5161.7 2158.79  5171.7 2160.37  5184.2 2160.49
#Mann=4,-1,0
  4853.3    0.07       0  4989.0    0.07       0  4993.0    0.07       0
  5020.7    0.16       0
Bank Sta=4989,4993
Exp/Cntr=0.3,0.1

Type RM Length L Ch R = 1,8091,70,70,70
BEGIN DESCRIPTION:
Elm 79 8091.19
END DESCRIPTION:
XS GIS Cut Line= 3
      1536012.68      6764344.78      1536153.31      6764363.87
      1536299.11      6764343.05
#Sta/Elev= 30
  4856.8 2132.55  4860.5 2132.55  4869.2 2131.70  4879.3 2131.22  4909.6 2128.47
  4916.3 2126.63  4921.3 2127.88  4929.8 2125.47  4939.9 2121.73  4960.1 2111.33
  4970.1 2108.44  4980.2 2108.48  4986.8 2108.00  4987.0 2107.50  4990.5 2107.50
  4990.8 2108.00  4993.8 2108.14  5001.8 2108.00  5010.5 2108.82  5020.6 2109.48
  5030.7 2112.50  5040.8 2117.52  5061.0 2126.81  5070.8 2131.87  5075.9 2131.81
  5081.2 2137.71  5101.4 2147.59  5111.5 2152.21  5121.6 2155.84  5146.0 2155.64
#Mann=3,-1,0
  4856.8    0.07       0  4986.8    0.07       0  4990.8    0.16       0
Bank Sta=4986.8,4990.8
Exp/Cntr=0.3,0.1

Type RM Length L Ch R = 1,8021,92,92,92
BEGIN DESCRIPTION:
Elm 79 8021.34
END DESCRIPTION:
XS GIS Cut Line= 3
      1536023.14      6764402.07      1536186.30      6764422.90
      1536311.54      6764402.31
#Sta/Elev= 30
  4832.8 2130.48  4836.2 2130.48  4839.9 2129.44  4845.0 2129.40  4864.9 2127.16
  4895.2 2125.62  4914.7 2120.49  4919.7 2119.60  4925.4 2116.52  4935.5 2112.76
  4945.6 2107.94  4963.0 2107.43  4963.7 2107.41  4964.0 2106.91  4967.5 2106.91
  4967.7 2107.41  5006.1 2107.98  5016.2 2108.86  5026.4 2110.58  5036.5 2113.88
  5046.6 2119.19  5055.0 2124.89  5060.1 2126.70  5066.9 2132.84  5077.0 2139.78
  5087.2 2148.62  5097.3 2155.72  5116.2 2154.80  5121.3 2155.22  5124.2 2155.09
#Mann=4,-1,0
  4832.8    0.07       0  4963.0    0.16       0  4963.7    0.07       0
  4967.7    0.16       0
Bank Sta=4963.7,4967.7
Exp/Cntr=0.3,0.1

Type RM Length L Ch R = 1,7929,98,98,98
BEGIN DESCRIPTION:
Elm 79 7929.03
END DESCRIPTION:
XS GIS Cut Line= 3
      1535988.42      6764466.31      1536158.52      6764499.29
      1536314.75      6764461.10
#Sta/Elev= 30
  4828.9 2131.25  4856.0 2129.50  4886.5 2125.36  4906.9 2121.05  4914.3 2117.30
  4919.4 2117.70  4937.5 2112.76  4957.8 2112.24  4971.1 2110.81  4986.4 2108.03
  4986.6 2107.53  4990.4 2108.03  5007.0 2108.26  5031.6 2110.39  5039.7 2109.65
  5060.3 2110.53  5068.1 2113.97  5073.3 2112.97  5091.2 2123.29  5101.5 2130.16
  5109.8 2136.60  5114.9 2137.39  5122.1 2144.64  5132.4 2148.52  5142.7 2147.52
  5151.4 2144.74  5156.6 2149.21  5160.6 2146.49  5161.9 2146.49  5163.0 2146.49
#Mann=5,-1,0
  4828.9    0.07       0  4986.4    0.07       0  4990.4    0.07       0
  5007.0    0.16       0  5161.9    0.07       0
Bank Sta=4986.4,4990.4
Exp/Cntr=0.3,0.1

Type RM Length L Ch R = 1,7831,101,101,101
BEGIN DESCRIPTION:
Elm 79 7831.43
END DESCRIPTION:
XS GIS Cut Line= 3
      1535941.56      6764568.74      1536155.05      6764596.51
      1536255.75      6764580.89
#Sta/Elev= 30
  4784.4 2130.43  4808.0 2128.92  4815.2 2127.95  4820.3 2128.44  4828.2 2126.68
  4868.5 2120.44  4888.7 2118.26  4894.3 2117.14  4899.4 2118.42  4908.9 2115.55
  4920.2 2112.97  4929.1 2112.01  4949.2 2106.18  4957.3 2105.02  4957.6 2104.52
  4961.1 2104.52  4961.3 2105.02  4989.6 2105.24  4997.1 2105.89  5009.8 2105.58
  5018.7 2106.52  5023.8 2106.38  5030.0 2111.41  5040.1 2117.77  5060.4 2128.93
  5080.6 2138.41  5086.7 2137.79  5091.8 2140.86  5098.7 2139.70  5101.6 2139.70
#Mann=4,-1,0
  4784.4    0.07       0  4920.2    0.16       0  4957.3    0.07       0
  4961.3    0.16       0
Bank Sta=4957.3,4961.3
Exp/Cntr=0.3,0.1

Type RM Length L Ch R = 1,7730,72,72,72
BEGIN DESCRIPTION:
Elm 79 7729.89
END DESCRIPTION:
XS GIS Cut Line= 3
      1536000.51      6764626.01      1536104.70      6764685.05
      1536309.57      6764657.28
#Sta/Elev= 30
  4872.1 2127.19  4877.6 2127.19  4884.6 2124.75  4890.4 2124.93  4906.3 2121.21
  4912.0 2121.12  4922.2 2118.21  4927.9 2117.98  4943.8 2111.53  4949.5 2111.15
  4956.5 2106.57  4965.4 2104.19  4971.2 2103.72  5000.2 2103.47  5000.4 2102.97
  5004.2 2103.47  5042.6 2104.94  5062.8 2109.79  5072.9 2110.54  5093.1 2114.04
  5103.2 2114.05  5113.3 2111.39  5123.3 2107.52  5133.4 2107.38  5152.3 2111.05
  5157.3 2108.49  5160.7 2109.31  5173.8 2114.14  5193.8 2124.80  5198.6 2124.80
#Mann=5,-1,0
  4872.1    0.07       0  4956.5    0.16       0  5000.2    0.07       0
  5004.2    0.16       0  5160.7    0.07       0
Bank Sta=5000.2,5004.2
Exp/Cntr=0.3,0.1

Type RM Length L Ch R = 1,7658,78,78,78
BEGIN DESCRIPTION:
Elm 79 7658.4
END DESCRIPTION:
XS GIS Cut Line= 3
      1535948.49      6764686.81      1536106.44      6764754.50
      1536276.57      6764778.80
#Sta/Elev= 30
  4829.4 2128.25  4843.5 2126.00  4857.3 2125.16  4872.5 2123.59  4890.7 2123.21
  4912.6 2119.88  4934.4 2115.04  4943.3 2112.10  4948.7 2112.47  4956.2 2108.43
  4966.8 2105.13  4972.3 2104.74  4977.9 2101.45  4986.8 2100.74  4987.0 2100.24
  4990.5 2100.24  4990.8 2100.74  5030.1 2101.31  5050.3 2103.42  5063.4 2103.07
  5070.5 2106.79  5080.6 2110.34  5100.8 2119.23  5121.0 2130.18  5129.1 2135.63
  5134.1 2136.55  5141.2 2141.36  5151.3 2145.52  5165.3 2148.77  5173.1 2149.52
#Mann=5,-1,0
  4829.4    0.07       0  4857.3    0.16       0  4986.8    0.07       0
  4990.8    0.16       0  5165.3    0.07       0
Bank Sta=4986.8,4990.8
Exp/Cntr=0.3,0.1

Type RM Length L Ch R = 1,7580,133,133,133
BEGIN DESCRIPTION:
Elm 79 7580.306
END DESCRIPTION:
XS GIS Cut Line= 3
      1535904.98      6764788.00      1536102.73      6764832.06
      1536255.02      6764838.00
#Sta/Elev= 30
  4797.4 2138.79  4800.0 2138.79  4807.7 2136.12  4816.6 2131.67  4821.7 2131.85
  4824.9 2130.46  4838.4 2126.10  4848.6 2124.22  4865.2 2119.51  4879.4 2119.44
  4889.6 2117.80  4913.8 2111.90  4920.4 2108.84  4930.6 2105.44  4957.3 2099.46
  4996.6 2098.50  4996.9 2098.00  5000.4 2098.00  5000.6 2098.50  5012.3 2099.16
  5025.7 2100.94  5032.3 2103.86  5052.3 2106.70  5062.3 2108.83  5082.3 2114.63
  5092.3 2118.70  5122.4 2133.71  5142.4 2145.03  5149.9 2148.19  5152.4 2148.19
#Mann=4,-1,0
  4797.4    0.07       0  4824.9    0.16       0  4996.6    0.07       0
  5000.6    0.16       0
Bank Sta=4996.6,5000.6
Exp/Cntr=0.3,0.1

Type RM Length L Ch R = 1,7447,179,179,179
BEGIN DESCRIPTION:
Elm 79 7446.7
END DESCRIPTION:
XS GIS Cut Line= 3
      1535927.66      6764888.20      1536059.56      6764952.42
      1536217.55      6764952.42
#Sta/Elev= 30
  4858.8 2123.82  4871.2 2119.34  4878.1 2117.39  4888.1 2115.84  4903.9 2114.49
  4916.2 2113.10  4922.6 2109.00  4933.2 2104.25  4938.8 2102.76  4944.8 2098.12
  4967.1 2093.21  4978.2 2092.84  4989.4 2091.84  4998.2 2091.77  4998.4 2091.27
  5001.9 2091.27  5002.2 2091.77  5010.9 2091.88  5020.9 2093.13  5030.9 2097.95
  5040.9 2101.09  5060.9 2104.67  5070.9 2107.15  5080.9 2111.09  5090.9 2113.09
  5100.9 2116.74  5120.9 2123.32  5130.9 2126.00  5159.7 2135.28  5163.5 2135.28
#Mann=4,-1,0
  4858.8    0.07       0  4903.9    0.16       0  4998.2    0.07       0
  5002.2    0.16       0
Bank Sta=4998.2,5002.2
Exp/Cntr=0.3,0.1

Type RM Length L Ch R = 1,7268,165,165,165
BEGIN DESCRIPTION:
Elm 79 7268.18
END DESCRIPTION:
XS GIS Cut Line= 3
      1535880.74      6764863.86      1535991.86      6765103.46
      1536129.00      6765242.34
#Sta/Elev= 30
  4737.1 2129.06  4804.5 2117.36  4850.3 2115.13  4907.1 2106.12  4936.0 2105.53
  4952.9 2103.43  4964.2 2106.21  4970.3 2107.62  4975.8 2104.42  5007.0 2108.16
  5013.7 2104.93  5020.8 2106.87  5027.9 2104.46  5049.1 2107.51  5075.4 2098.31
  5075.7 2097.81  5079.4 2098.31  5091.5 2099.70  5098.6 2105.20  5105.7 2101.76
  5119.8 2108.40  5126.9 2108.31  5134.0 2114.63  5141.0 2112.69  5148.1 2118.87
  5155.1 2117.10  5169.3 2125.25  5176.3 2125.02  5183.4 2129.39  5196.4 2128.51
#Mann=5,-1,0
  4737.1    0.07       0  4936.0    0.16       0  4964.2    0.07       0
  5075.4    0.07       0  5079.4    0.07       0
Bank Sta=5075.4,5079.4
Exp/Cntr=0.3,0.1

Type RM Length L Ch R = 1,7103,49,49,49
BEGIN DESCRIPTION:
Elm 79 7103.395
END DESCRIPTION:
XS GIS Cut Line= 3
      1535705.03      6765088.02      1535908.76      6765239.56
      1536055.04      6765288.01
#Sta/Elev= 30
  4746.1 2136.96  4749.2 2136.96  4753.4 2134.76  4774.2 2128.09  4788.8 2125.84
  4803.4 2121.80  4826.2 2118.34  4832.6 2116.50  4838.9 2115.93  4853.5 2111.77
  4874.3 2107.93  4895.6 2101.68  4924.4 2097.00  4945.5 2091.23  4953.6 2092.54
  4968.2 2093.08  4994.5 2090.55  5035.8 2089.89  5036.1 2089.39  5039.8 2089.89
  5048.7 2094.27  5074.8 2103.87  5080.3 2107.65  5086.4 2109.95  5106.5 2116.94
  5111.9 2121.50  5132.9 2130.53  5138.2 2131.83  5143.5 2135.16  5154.1 2136.55
#Mann=5,-1,0
  4746.1    0.07       0  4826.2    0.16       0  5035.8    0.07       0
  5039.8    0.16       0  5086.4    0.07       0
Bank Sta=5035.8,5039.8
Exp/Cntr=0.3,0.1

Type RM Length L Ch R = 1,7054,65,65,65
BEGIN DESCRIPTION:
Elm 79 7053.69
END DESCRIPTION:
XS GIS Cut Line= 3
      1535668.92      6765155.53      1535908.52      6765290.96
      1536057.81      6765337.83
#Sta/Elev= 30
  4728.9 2130.59  4742.9 2129.27  4748.6 2127.43  4758.8 2126.91  4786.1 2121.13
  4795.4 2117.69  4839.3 2106.14  4873.7 2098.88  4882.9 2096.14  4888.6 2092.68
  4896.7 2091.73  4904.6 2093.49  4919.7 2090.30  4963.8 2090.67  4997.2 2088.75
  4997.5 2088.25  5001.2 2088.75  5021.4 2089.41  5040.7 2098.21  5046.0 2099.63
  5052.8 2104.44  5073.1 2109.66  5078.4 2109.82  5084.3 2113.52  5097.8 2118.19
  5105.2 2120.99  5110.8 2125.28  5116.0 2126.20  5143.2 2136.09  5160.6 2136.44
#Mann=5,-1,0
  4728.9    0.07       0  4795.4    0.16       0  4997.2    0.07       0
  5001.2    0.16       0  5097.8    0.07       0
Bank Sta=4997.2,5001.2
Exp/Cntr=0.3,0.1

Type RM Length L Ch R = 1,6989,45,45,45
BEGIN DESCRIPTION:
Elm 79 6989.13
END DESCRIPTION:
XS GIS Cut Line= 3
      1535674.13      6765219.77      1535905.05      6765353.46
      1536061.53      6765380.97
#Sta/Elev= 30
  4733.0 2118.75  4736.2 2118.75  4739.6 2116.71  4755.8 2118.58  4761.1 2116.08
  4768.7 2116.28  4776.9 2114.91  4782.7 2111.32  4798.4 2106.51  4804.2 2102.76
  4814.2 2100.63  4820.0 2096.24  4826.4 2093.40  4841.5 2090.13  4863.0 2088.71
  4943.4 2088.81  4974.9 2090.53  4988.2 2087.42  4997.4 2086.75  4997.6 2086.25
  5001.4 2086.75  5009.9 2088.06  5030.2 2101.98  5050.2 2107.42  5055.3 2105.75
  5060.7 2109.41  5101.4 2124.99  5121.6 2132.71  5131.8 2134.27  5158.7 2135.68
#Mann=5,-1,0
  4733.0    0.07       0  4755.8    0.16       0  4997.4    0.07       0
  5001.4    0.16       0  5101.4    0.07       0
Bank Sta=4997.4,5001.4
Exp/Cntr=0.3,0.1

Type RM Length L Ch R = 1,6944,83,83,83
BEGIN DESCRIPTION:
Elm 79 6943.94
END DESCRIPTION:
XS GIS Cut Line= 3
      1535627.31      6765336.10      1535898.11      6765396.86
      1536070.82      6765414.13
#Sta/Elev= 30
  4726.3 2140.46  4745.3 2129.07  4753.7 2122.25  4758.8 2124.98  4764.9 2118.69
  4795.7 2097.32  4802.1 2090.75  4807.3 2090.62  4816.2 2087.09  4845.5 2086.91
  4850.6 2086.18  4867.4 2087.52  4899.1 2087.35  4928.9 2088.96  4959.6 2088.80
  4978.1 2085.43  4978.4 2084.93  4982.1 2085.43  5003.8 2086.26  5010.8 2089.12
  5020.8 2091.19  5040.9 2097.59  5060.8 2106.06  5065.8 2105.63  5071.1 2109.41
  5101.2 2119.21  5116.4 2125.49  5141.4 2133.87  5161.3 2134.21  5177.4 2133.25
#Mann=5,-1,0
  4726.3    0.07       0  4745.3    0.16       0  4978.1    0.07       0
  4982.1    0.16       0  5116.4    0.07       0
Bank Sta=4978.1,4982.1
Exp/Cntr=0.3,0.1

Type RM Length L Ch R = 1,6861,64,64,64
BEGIN DESCRIPTION:
Elm 79 6860.7
END DESCRIPTION:
XS GIS Cut Line= 3
      1535658.51      6765386.44      1535840.81      6765457.62
      1536097.74      6765533.49
#Sta/Elev= 30
  4808.4 2134.42  4815.4 2125.88  4823.6 2118.36  4829.0 2120.27  4836.8 2112.48
  4847.6 2105.36  4853.4 2098.91  4858.8 2101.84  4877.9 2087.63  4883.3 2088.98
  4890.5 2086.03  4901.3 2085.59  4986.6 2086.51  5001.7 2083.56  5001.9 2083.06
  5005.7 2083.56  5056.9 2089.10  5062.1 2088.68  5090.2 2092.81  5102.3 2092.43
  5123.2 2095.40  5162.0 2104.26  5195.5 2113.67  5200.5 2115.45  5217.0 2124.54
  5227.4 2126.95  5233.8 2130.23  5248.3 2130.87  5258.7 2127.73  5272.0 2127.55
#Mann=4,-1,0
  4808.4    0.16       0  5001.7    0.07       0  5005.7    0.16       0
  5195.5    0.07       0
Bank Sta=5001.7,5005.7
Exp/Cntr=0.3,0.1

Type RM Length L Ch R = 1,6797,100,100,100
BEGIN DESCRIPTION:
Elm 79 6797.3
END DESCRIPTION:
XS GIS Cut Line= 3
      1535644.63      6765414.22      1535816.51      6765514.92
      1536076.96      6765554.85
#Sta/Elev= 30
  4813.9 2136.51  4825.7 2136.73  4831.5 2133.48  4847.2 2127.88  4853.0 2123.29
  4860.7 2120.34  4868.7 2115.31  4874.5 2115.31  4883.9 2110.60  4890.1 2104.13
  4895.9 2104.49  4905.8 2097.89  4911.6 2099.98  4927.3 2088.47  4933.1 2089.58
  4941.8 2084.69  5011.2 2083.80  5029.8 2082.17  5030.1 2081.67  5033.8 2082.17
  5163.3 2094.16  5193.5 2102.19  5198.6 2099.32  5203.8 2102.41  5228.3 2111.49
  5254.4 2119.39  5261.9 2122.93  5267.0 2119.83  5273.1 2126.52  5276.6 2126.52
#Mann=4,-1,0
  4813.9    0.16       0  5029.8    0.07       0  5033.8    0.16       0
  5228.3    0.07       0
Bank Sta=5029.8,5033.8
Exp/Cntr=0.3,0.1

Type RM Length L Ch R = 1,6697,57,57,57
BEGIN DESCRIPTION:
Elm 79 6696.64
END DESCRIPTION:
XS GIS Cut Line= 3
      1535665.44      6765440.24      1535804.36      6765580.89
      1536011.32      6765651.60
#Sta/Elev= 30
  4760.0 2126.31  4772.2 2119.96  4828.8 2104.54  4835.9 2102.16  4842.9 2097.79
  4857.1 2092.79  4864.2 2094.68  4871.2 2092.62  4878.3 2094.02  4885.4 2091.62
  4892.5 2092.84  4899.5 2090.22  4906.6 2090.42  4913.6 2087.16  4920.8 2086.74
  4927.8 2084.18  4960.7 2082.98  4963.9 2081.45  4993.2 2080.20  4993.5 2079.70
  4997.2 2080.20  5000.6 2081.81  5074.6 2084.76  5089.2 2091.27  5095.7 2096.01
  5115.2 2102.74  5146.8 2117.89  5159.1 2125.15  5169.7 2126.00  5176.4 2123.31
#Mann=4,-1,0
  4760.0    0.16       0  4993.2    0.07       0  4997.2    0.16       0
  5146.8    0.07       0
Bank Sta=4993.2,4997.2
Exp/Cntr=0.3,0.1

Type RM Length L Ch R = 1,6640,90,90,90
BEGIN DESCRIPTION:
Elm 79 6639.588
END DESCRIPTION:
XS GIS Cut Line= 3
      1535654.99      6765437.98      1535809.42      6765639.64
      1535955.00      6765688.00
#Sta/Elev= 30
  4746.0 2129.35  4749.2 2129.35  4753.3 2125.53  4767.8 2121.07  4774.1 2117.90
  4838.5 2100.30  4846.7 2099.82  4853.0 2097.25  4859.4 2097.49  4888.3 2094.67
  4923.7 2087.98  4938.2 2086.77  4960.1 2087.38  4967.2 2086.74  4973.5 2082.93
  5000.0 2081.72  5008.9 2079.49  5009.2 2078.99  5012.9 2079.49  5037.3 2082.08
  5042.6 2081.41  5074.2 2082.66  5079.6 2086.38  5100.6 2096.38  5121.8 2110.58
  5132.3 2114.12  5142.9 2123.46  5146.6 2124.97  5150.8 2126.69  5153.4 2126.69
#Mann=4,-1,0
  4746.0    0.16       0  5008.9    0.07       0  5012.9    0.16       0
  5146.6    0.07       0
Bank Sta=5008.9,5012.9
Exp/Cntr=0.3,0.1

Type RM Length L Ch R = 1,6550,116,116,116
BEGIN DESCRIPTION:
Elm 79 6550.01
END DESCRIPTION:
XS GIS Cut Line= 3
      1535599.48      6765520.11      1535776.58      6765721.51
      1535920.33      6765818.50
#Sta/Elev= 30
  4734.6 2119.43  4736.9 2116.81  4751.1 2113.32  4779.6 2099.01  4793.8 2094.78
  4871.6 2087.40  4900.1 2085.44  4906.8 2085.98  4949.5 2080.94  4971.3 2080.41
  4977.9 2078.63  4990.1 2077.80  4990.4 2077.30  4994.1 2077.80  5027.2 2079.81
  5042.2 2081.93  5057.1 2088.33  5063.2 2092.06  5072.1 2094.70  5085.3 2100.86
  5093.1 2102.77  5099.1 2107.24  5108.1 2108.24  5114.1 2113.91  5115.7 2114.20
  5129.1 2118.03  5135.1 2123.86  5144.1 2126.28  5150.1 2130.97  5176.2 2129.62
#Mann=4,-1,0
  4734.6    0.16       0  4990.1    0.07       0  4994.1    0.16       0
  5115.7    0.07       0
Bank Sta=4990.1,4994.1
Exp/Cntr=0.3,0.1

Type RM Length L Ch R = 1,6434,113,113,113
BEGIN DESCRIPTION:
Elm 79 6434.36
END DESCRIPTION:
XS GIS Cut Line= 3
      1535545.70      6765560.09      1535726.23      6765822.21
      1535847.75      6765867.34
#Sta/Elev= 30
  4685.2 2116.65  4690.8 2111.59  4696.8 2109.83  4705.6 2104.23  4711.7 2102.23
  4719.1 2097.43  4726.6 2093.88  4762.4 2084.34  4783.4 2083.86  4813.2 2080.96
  4834.1 2081.68  4849.0 2079.81  4855.1 2080.66  4920.7 2077.63  4941.7 2078.85
  4956.5 2077.24  4962.6 2078.16  4990.4 2076.84  4990.6 2076.34  4994.4 2076.84
  5031.7 2078.06  5044.8 2083.33  5055.5 2086.02  5087.0 2106.01  5092.4 2117.39
  5097.5 2125.86  5098.2 2127.02  5117.4 2128.28  5122.7 2129.66  5133.1 2129.42
#Mann=4,-1,0
  4685.2    0.16       0  4990.4    0.07       0  4994.4    0.16       0
  5097.5    0.07       0
Bank Sta=4990.4,4994.4
Exp/Cntr=0.3,0.1

Type RM Length L Ch R = 1,6321,102,102,102
BEGIN DESCRIPTION:
Elm 79 6320.79
END DESCRIPTION:
XS GIS Cut Line= 3
      1535446.75      6765603.49      1535661.99      6765846.51
      1535856.48      6765891.66
#Sta/Elev= 30
  4720.8 2127.94  4737.1 2122.70  4743.8 2117.22  4751.4 2116.23  4758.0 2111.04
  4765.6 2109.74  4786.5 2098.34  4800.7 2095.05  4821.6 2084.51  4835.8 2080.96
  4878.5 2077.80  4970.5 2077.23  4990.3 2074.55  4990.5 2074.05  4994.3 2074.55
  5027.4 2076.06  5043.9 2082.96  5069.0 2080.46  5074.2 2086.09  5099.9 2084.30
  5116.8 2087.13  5121.9 2093.06  5159.4 2101.88  5164.6 2108.29  5183.4 2117.13
  5192.2 2125.21  5202.1 2128.05  5207.2 2123.64  5223.0 2128.54  5245.1 2129.39
#Mann=4,-1,0
  4720.8    0.16       0  4990.3    0.07       0  4994.3    0.16       0
  5183.4    0.07       0
Bank Sta=4990.3,4994.3
Exp/Cntr=0.3,0.1
