HEC-RAS study Elm 79.prj: Elm 79 Base Level Engineering

--- Elm 79.g01 (geometry) --- (continued)

Type RM Length L Ch R = 1,6219,169,169,169
BEGIN DESCRIPTION:
Elm 79 6219.35
END DESCRIPTION:
XS GIS Cut Line= 3
      1535323.48      6765704.17      1535563.04      6765886.44
      1535871.05      6765917.59
#Sta/Elev= 30
  4700.8 2124.02  4712.2 2123.90  4718.5 2120.77  4724.4 2120.38  4747.6 2114.68
  4753.8 2111.23  4762.1 2109.92  4790.7 2098.67  4803.7 2092.09  4832.8 2082.82
  4868.2 2080.12  4903.8 2075.94  4976.2 2074.69  4997.9 2068.61  4998.2 2068.11
  5001.9 2068.61  5013.8 2068.93  5084.2 2086.15  5114.4 2090.73  5134.5 2097.04
  5163.0 2102.90  5168.0 2099.54  5174.7 2101.33  5184.7 2101.49  5216.6 2106.97
  5245.0 2111.58  5262.9 2116.53  5268.0 2111.86  5295.3 2119.32  5311.4 2121.98
#Mann=5,-1,0
  4700.8    0.07       0  4724.4    0.16       0  4997.9    0.07       0
  5001.9    0.16       0  5216.6    0.07       0
Bank Sta=4997.9,5001.9
Exp/Cntr=0.3,0.1

Type RM Length L Ch R = 1,6050,194,194,194
BEGIN DESCRIPTION:
Elm 79 6050.17
END DESCRIPTION:
XS GIS Cut Line= 3
      1535276.56      6765877.75      1535448.45      6765990.61
      1535767.86      6766087.82
#Sta/Elev= 30
  4786.6 2116.42  4814.5 2108.75  4829.6 2099.53  4835.6 2098.55  4844.5 2093.84
  4850.7 2088.56  4856.7 2087.43  4865.8 2082.39  4890.6 2079.57  4974.3 2073.05
  5002.4 2074.40  5028.0 2072.00  5028.2 2071.50  5032.0 2072.00  5040.9 2074.19
  5068.1 2072.95  5073.3 2075.15  5124.5 2075.82  5133.8 2076.66  5139.0 2079.63
  5171.9 2081.40  5177.1 2079.69  5204.7 2082.20  5209.9 2080.79  5237.6 2082.34
  5242.8 2080.96  5270.4 2092.25  5276.3 2092.10  5281.3 2096.72  5326.1 2109.73
#Mann=5,-1,0
  4786.6    0.07       0  4890.6    0.16       0  5028.0    0.07       0
  5032.0    0.16       0  5276.3    0.07       0
Bank Sta=5028,5032
Exp/Cntr=0.3,0.1

Type RM Length L Ch R = 1,5856,259,259,259
BEGIN DESCRIPTION:
Elm 79 5855.92
END DESCRIPTION:
XS GIS Cut Line= 3
      1535288.73      6766202.41      1535542.20      6766108.67
      1535759.25      6766138.18
#Sta/Elev= 30
  4780.4 2092.08  4805.3 2087.53  4810.6 2088.19  4835.7 2082.40  4841.0 2083.43
  4860.8 2079.21  4866.1 2081.21  4872.4 2078.70  4883.0 2076.73  4915.0 2074.21
  4921.6 2072.09  4926.9 2072.82  4977.1 2069.54  5000.3 2066.67  5005.4 2065.18
  5005.7 2064.68  5009.5 2065.18  5012.8 2065.27  5021.6 2069.16  5032.3 2070.90
  5144.3 2074.40  5153.2 2075.95  5158.2 2074.92  5174.6 2077.97  5204.9 2084.66
  5225.0 2091.46  5230.7 2098.38  5235.7 2099.28  5265.0 2114.63  5269.7 2114.63
#Mann=3,-1,0
  4780.4    0.16       0  5005.4    0.07       0  5009.5    0.16       0
Bank Sta=5005.4,5009.5
Exp/Cntr=0.3,0.1

Type RM Length L Ch R = 1,5597,246,246,246
BEGIN DESCRIPTION:
Elm 79 5596.78
END DESCRIPTION:
XS GIS Cut Line= 3
      1535259.21      6766280.54      1535604.70      6766311.79
      1535761.35      6766318.68
#Sta/Elev= 30
  4652.9 2090.28  4658.7 2088.56  4668.8 2087.20  4677.0 2087.44  4682.0 2085.61
  4688.8 2085.43  4698.9 2083.19  4729.0 2079.94  4799.3 2068.77  4819.4 2067.91
  4889.7 2068.37  4903.5 2067.47  4909.7 2064.05  4919.8 2067.56  4949.9 2067.53
  4959.9 2066.36  4970.0 2062.68  4978.0 2062.33  4978.2 2061.83  4982.1 2062.33
  4990.1 2068.71  4997.4 2073.07  5002.5 2073.07  5010.1 2076.08  5040.1 2082.38
  5070.2 2092.21  5090.2 2101.79  5110.2 2114.01  5125.9 2118.98  5156.6 2128.03
#Mann=4,-1,0
  4652.9    0.16       0  4978.0    0.07       0  4982.1    0.16       0
  5125.9    0.07       0
Bank Sta=4978,4982.1
Exp/Cntr=0.3,0.1

Type RM Length L Ch R = 1,5351,153,153,153
BEGIN DESCRIPTION:
Elm 79 5351.05
END DESCRIPTION:
XS GIS Cut Line= 3
      1535203.63      6766306.56      1535441.51      6766494.08
      1535675.92      6766542.70
#Sta/Elev= 30
  4689.6 2094.43  4719.7 2090.36  4727.7 2086.73  4734.1 2086.91  4763.0 2083.52
  4769.4 2081.25  4805.9 2073.57  4862.4 2066.76  4905.7 2064.25  4976.2 2064.28
  4984.2 2063.16  4990.7 2059.47  5014.4 2057.77  5014.7 2057.27  5018.5 2057.77
  5026.7 2058.75  5034.1 2063.11  5039.2 2063.96  5108.4 2065.12  5118.6 2065.74
  5134.4 2069.72  5139.5 2069.20  5159.5 2078.68  5179.5 2090.12  5184.6 2089.72
  5190.1 2096.51  5210.5 2109.79  5220.7 2118.90  5228.9 2123.82  5231.9 2123.82
#Mann=3,-1,0
  4689.6    0.16       0  5014.4    0.07       0  5018.5    0.16       0
Bank Sta=5014.4,5018.5
Exp/Cntr=0.3,0.1

Type RM Length L Ch R = 1,5198,142,142,142
BEGIN DESCRIPTION:
Elm 79 5198.259
END DESCRIPTION:
XS GIS Cut Line= 3
      1535055.03      6766238.03      1535402.92      6766632.29
      1535555.04      6766688.01
#Sta/Elev= 30
  4474.2 2115.81  4502.2 2112.16  4538.2 2100.40  4566.6 2095.24  4630.2 2094.10
  4658.6 2088.27  4679.5 2087.83  4687.1 2086.12  4693.8 2087.03  4708.0 2082.39
  4728.9 2080.39  4764.9 2073.00  4800.0 2062.24  4941.4 2061.21  4967.8 2056.34
  4968.0 2055.84  4971.9 2056.34  4977.4 2056.41  4984.0 2059.35  5004.8 2059.59
  5035.3 2062.84  5060.5 2072.44  5066.1 2076.55  5085.7 2084.30  5116.2 2092.95
  5121.5 2096.62  5130.0 2099.32  5146.7 2102.97  5152.0 2107.37  5162.0 2107.68
#Mann=3,-1,0
  4474.2    0.16       0  4967.8    0.07       0  4971.9    0.16       0
Bank Sta=4967.8,4971.9
Exp/Cntr=0.3,0.1

Type RM Length L Ch R = 1,5056,161,161,161
BEGIN DESCRIPTION:
Elm 79 5056.29
END DESCRIPTION:
XS GIS Cut Line= 3
      1535139.45      6766468.07      1535288.73      6766704.15
      1535420.31      6766920.57
#Sta/Elev= 30
  4720.0 2090.31  4759.9 2076.56  4775.2 2074.25  4781.1 2075.01  4802.7 2071.06
  4811.6 2070.52  4817.5 2072.01  4832.8 2069.19  4854.0 2068.79  4905.7 2064.99
  4921.0 2062.92  4932.9 2058.52  4998.6 2058.78  5005.7 2058.04  5019.1 2054.07
  5019.4 2053.57  5023.2 2054.07  5027.2 2057.26  5042.5 2060.47  5058.0 2060.23
  5085.7 2062.30  5109.2 2065.68  5137.5 2071.74  5167.7 2080.97  5189.7 2090.39
  5202.8 2097.82  5211.1 2100.78  5216.9 2104.66  5238.2 2113.03  5252.6 2112.94
#Mann=3,-1,0
  4720.0    0.16       0  5019.1    0.07       0  5023.2    0.16       0
Bank Sta=5019.1,5023.2
Exp/Cntr=0.3,0.1

Type RM Length L Ch R = 1,4895,126,126,126
BEGIN DESCRIPTION:
Elm 79 4894.9
END DESCRIPTION:
XS GIS Cut Line= 3
      1534958.87      6766610.40      1535193.24      6766827.42
      1535310.65      6766931.01
#Sta/Elev= 30
  4673.4 2071.13  4676.1 2073.35  4697.1 2074.58  4711.2 2072.86  4747.0 2064.17
  4796.3 2057.07  4902.3 2054.99  4966.4 2056.30  4985.3 2052.02  4985.6 2051.52
  4989.4 2052.02  4990.6 2053.99  4997.0 2053.99  5001.5 2056.60  5030.0 2058.33
  5036.7 2062.00  5044.2 2061.66  5050.9 2066.02  5058.4 2066.06  5065.1 2071.01
  5072.7 2072.16  5079.3 2077.32  5086.9 2077.64  5093.6 2083.83  5101.1 2084.04
  5107.8 2088.97  5122.0 2091.18  5128.7 2095.93  5136.2 2097.51  5149.4 2103.50
#Mann=3,-1,0
  4673.4    0.16       0  4985.3    0.07       0  4989.4    0.16       0
Bank Sta=4985.3,4989.4
Exp/Cntr=0.3,0.1

Type RM Length L Ch R = 1,4769,125,125,125
BEGIN DESCRIPTION:
Elm 79 4769.174
END DESCRIPTION:
XS GIS Cut Line= 3
      1534804.98      6766787.99      1535081.44      6766860.86
      1535254.97      6766937.99
#Sta/Elev= 30
  4714.1 2091.59  4716.7 2091.59  4731.7 2085.17  4755.5 2078.37  4765.8 2076.99
  4772.0 2074.65  4810.8 2070.32  4847.4 2067.29  4887.7 2059.15  4928.0 2055.20
  4952.0 2053.97  5002.6 2054.02  5023.0 2052.16  5023.3 2051.66  5027.2 2052.16
  5053.8 2059.02  5069.6 2061.79  5077.1 2063.73  5082.6 2066.46  5100.3 2069.29
  5105.8 2072.49  5123.6 2076.33  5129.1 2079.48  5146.2 2084.26  5152.3 2086.66
  5157.8 2090.52  5175.6 2095.10  5181.0 2098.95  5187.2 2100.93  5189.9 2100.93
#Mann=4,-1,0
  4714.1    0.07       0  4810.8    0.16       0  5023.0    0.07       0
  5027.2    0.16       0
Bank Sta=5023,5027.2
Exp/Cntr=0.3,0.1

Type RM Length L Ch R = 1,4644,102,102,102
BEGIN DESCRIPTION:
Elm 79 4644.41
END DESCRIPTION:
XS GIS Cut Line= 3
      1534712.33      6766909.01      1535004.01      6766955.89
      1535260.74      6767062.72
#Sta/Elev= 30
  4703.2 2100.50  4707.1 2100.50  4724.7 2095.05  4729.8 2096.28  4776.8 2080.42
  4786.6 2077.56  4791.7 2077.43  4797.1 2073.28  4807.2 2070.07  4817.3 2068.73
  4827.4 2064.61  4837.6 2062.70  4853.6 2069.73  4857.7 2067.79  4898.3 2065.26
  4915.5 2065.50  4949.0 2060.58  4982.4 2053.01  5008.4 2051.73  5008.7 2051.23
  5012.6 2051.73  5069.7 2052.80  5170.5 2064.45  5175.9 2066.54  5194.3 2069.87
  5205.5 2075.69  5247.4 2091.17  5259.6 2097.35  5270.5 2101.05  5276.7 2104.79
#Mann=4,-1,0
  4703.2    0.07       0  4857.7    0.16       0  5008.4    0.07       0
  5012.6    0.16       0
Bank Sta=5008.4,5012.6
Exp/Cntr=0.3,0.1

Type RM Length L Ch R = 1,4542,98,98,98
BEGIN DESCRIPTION:
Elm 79 4541.68
END DESCRIPTION:
XS GIS Cut Line= 3
      1534741.84      6766948.94      1535007.48      6767060.05
      1535229.68      6767099.98
#Sta/Elev= 30
  4714.5 2094.84  4715.9 2094.84  4718.9 2094.84  4724.2 2091.58  4729.6 2090.66
  4771.8 2075.53  4815.5 2067.66  4837.0 2065.50  4848.0 2064.21  4854.0 2062.12
  4859.4 2063.86  4869.7 2062.83  4877.8 2057.36  4891.4 2054.56  4901.6 2055.26
  4930.8 2051.69  4976.0 2050.91  4976.3 2050.41  4980.2 2050.91  5060.9 2051.93
  5075.9 2052.91  5091.4 2056.32  5101.5 2056.38  5111.7 2058.44  5134.6 2064.89
  5142.2 2068.48  5172.6 2078.16  5213.3 2098.10  5223.3 2102.12  5228.2 2102.12
#Mann=5,-1,0
  4714.5    0.16       0  4715.9    0.07       0  4837.0    0.16       0
  4976.0    0.07       0  4980.2    0.16       0
Bank Sta=4976,4980.2
Exp/Cntr=0.3,0.1

Type RM Length L Ch R = 1,4444,152,152,152
BEGIN DESCRIPTION:
Elm 79 4443.94
END DESCRIPTION:
XS GIS Cut Line= 3
      1534701.92      6767068.73      1534957.13      6767141.65
      1535229.68      6767183.05
#Sta/Elev= 30
  4731.9 2097.58  4749.1 2094.83  4776.7 2086.67  4782.9 2082.17  4788.1 2082.50
  4807.9 2074.24  4821.9 2075.02  4828.7 2071.71  4855.7 2063.04  4874.3 2060.26
  4889.5 2055.60  4894.7 2057.00  4901.5 2054.50  4911.9 2053.03  4922.3 2053.65
  4953.5 2050.39  4982.6 2049.69  4982.9 2049.19  4986.8 2049.69  5025.5 2051.11
  5077.0 2051.10  5096.3 2056.00  5126.7 2058.01  5140.7 2060.51  5146.9 2063.22
  5187.3 2070.86  5209.4 2077.03  5248.0 2091.27  5267.9 2100.34  5273.0 2105.11
#Mann=4,-1,0
  4731.9    0.07       0  4874.3    0.16       0  4982.6    0.07       0
  4986.8    0.16       0
Bank Sta=4982.6,4986.8
Exp/Cntr=0.3,0.1

Type RM Length L Ch R = 1,4292,105,105,105
BEGIN DESCRIPTION:
Elm 79 4291.707
END DESCRIPTION:
XS GIS Cut Line= 3
      1534704.99      6767188.00      1534878.30      6767264.65
      1535254.96      6767238.00
#Sta/Elev= 30
  4810.5 2099.01  4816.5 2098.02  4822.9 2096.65  4848.2 2086.05  4854.2 2082.13
  4865.2 2082.06  4871.5 2077.77  4894.8 2067.47  4923.5 2058.13  4930.8 2054.69
  4936.3 2053.88  4952.7 2049.48  4970.1 2048.51  4973.4 2046.70  4973.7 2046.20
  4977.7 2046.70  4998.0 2048.92  5027.6 2049.80  5046.8 2048.10  5066.9 2048.39
  5197.2 2059.02  5207.2 2058.42  5227.3 2067.08  5277.4 2075.56  5297.4 2083.62
  5304.6 2087.95  5309.6 2088.63  5347.6 2104.59  5367.6 2110.81  5377.6 2111.33
#Mann=6,-1,0
  4810.5    0.07       0  4816.5    0.16       0  4822.9    0.07       0
  4936.3    0.16       0  4973.4    0.07       0  4977.7    0.16       0
Bank Sta=4973.4,4977.7
Exp/Cntr=0.3,0.1

Type RM Length L Ch R = 1,4187,148,148,148
BEGIN DESCRIPTION:
Elm 79 4186.7
END DESCRIPTION:
XS GIS Cut Line= 3
      1534663.70      6767228.43      1534809.56      6767343.04
      1535099.47      6767509.69
#Sta/Elev= 30
  4816.3 2095.21  4824.0 2093.68  4838.5 2093.98  4880.5 2083.72  4888.2 2078.68
  4902.6 2077.36  4914.7 2073.58  4923.4 2072.03  4931.5 2066.32  4937.9 2066.75
  4952.3 2059.59  4958.7 2059.11  4981.2 2049.61  5001.8 2046.31  5045.2 2047.59
  5058.8 2045.51  5059.1 2045.01  5063.1 2045.51  5125.7 2052.80  5141.5 2053.18
  5169.6 2057.42  5184.6 2057.07  5200.4 2061.61  5206.2 2059.82  5222.0 2062.78
  5227.7 2061.17  5265.1 2066.36  5273.4 2065.86  5308.2 2078.31  5336.2 2083.90
#Mann=5,-1,0
  4816.3    0.16       0  4880.5    0.07       0  4914.7    0.16       0
  5058.8    0.07       0  5063.1    0.16       0
Bank Sta=5058.8,5063.1
Exp/Cntr=0.3,0.1

Type RM Length L Ch R = 1,4039,97,97,97
BEGIN DESCRIPTION:
Elm 79 4038.95
END DESCRIPTION:
XS GIS Cut Line= 3
      1534462.34      6767405.54      1534807.83      6767490.61
      1535017.87      6767539.21
#Sta/Elev= 30
  4653.1 2089.25  4682.9 2084.32  4688.1 2086.18  4707.3 2082.63  4724.5 2080.76
  4729.6 2081.21  4758.8 2077.24  4805.5 2065.53  4841.2 2059.11  4849.0 2056.46
  4903.0 2048.55  4937.2 2045.96  4978.7 2046.06  4993.5 2042.73  4993.8 2042.23
  4997.8 2042.73  5004.9 2044.98  5015.3 2046.15  5047.1 2046.06  5057.3 2046.89
  5063.2 2048.57  5068.3 2047.95  5077.9 2050.07  5098.4 2051.66  5148.6 2063.01
  5160.0 2067.15  5190.8 2074.45  5201.5 2079.05  5211.3 2081.50  5224.5 2082.98
#Mann=4,-1,0
  4653.1    0.07       0  4805.5    0.16       0  4993.5    0.07       0
  4997.8    0.16       0
Bank Sta=4993.5,4997.8
Exp/Cntr=0.3,0.1

Type RM Length L Ch R = 1,3942,125,125,125
BEGIN DESCRIPTION:
Elm 79 3941.79
END DESCRIPTION:
XS GIS Cut Line= 3
      1534512.65      6767593.04      1534762.69      6767570.47
      1535045.70      6767587.83
#Sta/Elev= 30
  4755.1 2082.04  4759.0 2081.06  4787.6 2078.38  4803.9 2074.87  4818.7 2070.06
  4837.8 2063.31  4847.8 2061.18  4857.9 2057.29  4928.1 2045.66  4936.4 2045.16
  4975.7 2044.14  4980.7 2044.66  5009.8 2043.49  5016.3 2042.30  5016.6 2041.80
  5020.6 2042.30  5028.5 2044.12  5038.5 2044.99  5078.6 2044.78  5088.6 2045.89
  5098.6 2048.19  5118.7 2050.31  5128.7 2050.21  5158.8 2056.31  5198.8 2065.69
  5207.3 2068.35  5212.3 2066.88  5258.9 2084.27  5286.8 2091.64  5289.7 2091.64
#Mann=6,-1,0
  4755.1    0.07       0  4803.9    0.16       0  4818.7    0.07       0
  4936.4    0.16       0  5016.3    0.07       0  5020.6    0.16       0
Bank Sta=5016.3,5020.6
Exp/Cntr=0.3,0.1

Type RM Length L Ch R = 1,3817,244,244,244
BEGIN DESCRIPTION:
Elm 79 3817.334
END DESCRIPTION:
XS GIS Cut Line= 3
      1534505.01      6767738.00      1534746.85      6767694.06
      1535105.00      6767688.00
#Sta/Elev= 30
  4754.2 2095.65  4764.4 2093.07  4780.9 2085.84  4805.0 2081.54  4839.3 2072.33
  4845.7 2068.61  4866.0 2060.98  4876.2 2055.98  4886.3 2055.18  4892.7 2052.51
  4897.8 2052.27  4924.1 2046.33  4937.1 2042.99  4957.5 2043.47  4975.6 2040.02
  4975.9 2039.52  4979.9 2040.02  4996.5 2043.17  5088.2 2044.42  5108.2 2048.49
  5118.2 2049.23  5128.2 2047.59  5148.2 2052.83  5188.2 2057.36  5218.2 2065.01
  5268.2 2083.97  5298.2 2090.82  5328.2 2100.20  5338.2 2102.60  5358.2 2103.27
#Mann=4,-1,0
  4754.2    0.07       0  4924.1    0.16       0  4975.6    0.07       0
  4979.9    0.16       0
Bank Sta=4975.6,4979.9
Exp/Cntr=0.3,0.1

Type RM Length L Ch R = 1,3573,111,111,111
BEGIN DESCRIPTION:
Elm 79 3573.05
END DESCRIPTION:
XS GIS Cut Line= 3
      1534526.57      6767879.50      1534757.48      6767909.01
      1535089.07      6767797.90
#Sta/Elev= 30
  4770.9 2085.08  4801.6 2078.60  4829.8 2066.80  4850.0 2063.65  4881.8 2051.90
  4920.5 2041.22  4950.8 2040.54  4956.1 2038.75  4961.1 2040.11  4970.9 2039.49
  4978.9 2037.25  4979.2 2036.75  4983.2 2037.25  4999.9 2040.23  5056.6 2040.35
  5127.6 2045.44  5138.2 2046.85  5146.0 2050.02  5151.3 2047.82  5177.5 2053.65
  5182.8 2052.91  5214.4 2056.54  5264.7 2066.07  5272.2 2068.03  5277.5 2071.35
  5303.8 2075.17  5309.0 2079.20  5328.0 2081.73  5340.6 2086.77  5353.4 2088.78
#Mann=4,-1,0
  4770.9    0.07       0  4881.8    0.16       0  4978.9    0.07       0
  4983.2    0.16       0
Bank Sta=4978.9,4983.2
Exp/Cntr=0.3,0.1

Type RM Length L Ch R = 1,3462,139,139,139
BEGIN DESCRIPTION:
Elm 79 3461.51
END DESCRIPTION:
XS GIS Cut Line= 3
      1534512.74      6768013.18      1534755.74      6768020.12
      1535038.78      6767992.34
#Sta/Elev= 30
  4758.4 2065.27  4762.0 2065.27  4780.7 2061.78  4810.7 2058.39  4820.7 2055.49
  4851.7 2054.47  4880.7 2048.37  4900.7 2045.22  4920.7 2044.41  4930.7 2040.80
  4940.7 2039.13  4970.7 2039.22  4980.8 2037.91  4988.6 2035.48  4988.9 2034.98
  4992.9 2035.48  4998.6 2037.81  5003.6 2037.81  5010.8 2039.46  5075.3 2038.57
  5121.3 2040.92  5141.4 2043.51  5171.6 2049.31  5176.7 2051.47  5191.7 2055.16
  5211.8 2061.68  5252.0 2071.07  5278.1 2075.57  5282.5 2078.53  5285.9 2078.53
#Mann=4,-1,0
  4758.4    0.07       0  4851.7    0.16       0  4988.6    0.07       0
  4992.9    0.16       0
Bank Sta=4988.6,4992.9
Exp/Cntr=0.3,0.1

Type RM Length L Ch R = 1,3323,129,129,129
BEGIN DESCRIPTION:
Elm 79 3322.511
END DESCRIPTION:
XS GIS Cut Line= 3
      1534504.99      6768138.00      1534771.47      6768154.75
      1534955.01      6768138.00
#Sta/Elev= 30
  4733.0 2074.32  4743.0 2072.86  4753.0 2067.07  4763.1 2066.86  4773.1 2063.40
  4793.1 2058.37  4802.5 2056.82  4815.4 2055.07  4833.2 2055.43  4853.2 2054.05
  4873.3 2050.16  4883.3 2047.41  4933.4 2038.31  4993.5 2037.36  5004.3 2037.78
  5013.6 2036.86  5016.8 2034.24  5017.1 2033.74  5020.8 2033.74  5021.1 2034.24
  5024.0 2035.40  5033.7 2036.47  5063.8 2037.43  5083.9 2040.06  5093.9 2046.03
  5114.0 2054.36  5129.2 2066.79  5134.2 2065.17  5164.2 2074.29  5184.3 2077.15
#Mann=4,-1,0
  4733.0    0.07       0  4802.5    0.16       0  5016.8    0.07       0
  5021.1    0.16       0
Bank Sta=5016.8,5021.1
Exp/Cntr=0.3,0.1

Type RM Length L Ch R = 1,3194,110,110,110
BEGIN DESCRIPTION:
Elm 79 3193.96
END DESCRIPTION:
XS GIS Cut Line= 3
      1534521.35      6768174.63      1534852.97      6768251.03
      1535078.17      6768212.92
#Sta/Elev= 30
  4658.2 2069.49  4672.2 2067.79  4691.5 2060.98  4696.7 2060.40  4701.8 2058.68
  4733.8 2052.15  4764.6 2052.92  4774.8 2051.20  4782.3 2048.25  4787.4 2047.94
  4805.6 2041.94  4836.4 2036.93  4963.7 2036.54  4977.9 2033.22  4978.2 2032.72
  4982.2 2033.22  4990.3 2034.63  4997.0 2037.90  5002.1 2037.90  5020.8 2045.04
  5041.1 2050.85  5051.5 2055.83  5101.7 2060.94  5112.1 2064.80  5132.4 2067.71
  5162.1 2067.73  5167.2 2071.17  5203.4 2072.42  5222.5 2072.03  5226.9 2075.21
#Mann=4,-1,0
  4658.2    0.07       0  4701.8    0.16       0  4977.9    0.07       0
  4982.2    0.16       0
Bank Sta=4977.9,4982.2
Exp/Cntr=0.3,0.1

Type RM Length L Ch R = 1,3084,169,169,169
BEGIN DESCRIPTION:
Elm 79 3083.79
END DESCRIPTION:
XS GIS Cut Line= 3
      1534517.94      6768176.40      1534809.56      6768346.51
      1535200.08      6768339.57
#Sta/Elev= 30
  4664.7 2070.23  4678.2 2069.39  4684.5 2066.30  4713.1 2058.34  4752.7 2049.50
  4758.4 2049.00  4774.2 2050.86  4788.6 2049.43  4823.4 2040.63  4838.7 2038.83
  4846.5 2036.64  4993.3 2035.65  5002.3 2034.33  5005.6 2030.62  5005.9 2030.12
  5009.9 2030.62  5017.8 2033.89  5027.8 2035.26  5077.8 2038.45  5097.8 2043.16
  5117.8 2043.96  5157.8 2051.87  5196.3 2066.98  5201.3 2065.03  5207.8 2068.07
  5227.8 2071.57  5317.8 2074.66  5347.8 2076.64  5367.8 2076.22  5392.9 2073.87
#Mann=4,-1,0
  4664.7    0.07       0  4713.1    0.16       0  5005.6    0.07       0
  5009.9    0.16       0
Bank Sta=5005.6,5009.9
Exp/Cntr=0.3,0.1

Type RM Length L Ch R = 1,2915,90,90,90
BEGIN DESCRIPTION:
Elm 79 2915.44
END DESCRIPTION:
XS GIS Cut Line= 3
      1534509.22      6768186.79      1534811.30      6768520.12
      1535081.03      6768596.20
#Sta/Elev= 30
  4559.2 2074.22  4564.0 2069.73  4585.6 2067.83  4592.4 2064.25  4606.5 2060.13
  4622.2 2057.34  4641.8 2051.05  4663.3 2048.38  4670.1 2046.11  4748.5 2040.09
  4769.4 2037.10  4812.0 2034.73  4960.7 2033.15  4967.4 2031.00  4974.9 2032.28
  4981.6 2028.00  4986.9 2027.17  4987.2 2026.67  4991.2 2027.17  4995.8 2031.96
  5064.8 2032.91  5097.3 2037.53  5165.3 2065.85  5199.3 2074.76  5204.5 2072.27
  5231.1 2074.46  5256.3 2067.03  5262.3 2066.04  5272.5 2067.41  5289.3 2073.62
#Mann=5,-1,0
  4559.2    0.07       0  4622.2    0.16       0  4986.9    0.07       0
  4991.2    0.16       0  5256.3    0.07       0
Bank Sta=4986.9,4991.2
Exp/Cntr=0.3,0.1

Type RM Length L Ch R = 1,2825,158,158,158
BEGIN DESCRIPTION:
Elm 79 2824.903
END DESCRIPTION:
XS GIS Cut Line= 3
      1534454.99      6768187.98      1534756.35      6768586.21
      1535054.99      6768737.99
#Sta/Elev= 30
  4500.6 2076.50  4514.2 2077.96  4537.0 2076.30  4587.0 2067.94  4614.0 2060.29
  4635.0 2056.83  4678.5 2046.71  4713.9 2041.68  4751.3 2041.12  4807.5 2036.30
  4822.1 2036.96  4828.4 2034.64  4836.6 2036.29  4878.3 2032.87  4951.1 2030.79
  5002.0 2031.43  5018.7 2027.95  5019.0 2027.45  5023.1 2027.95  5031.8 2031.87
  5104.2 2032.05  5155.5 2040.08  5187.6 2043.13  5209.8 2053.04  5222.8 2061.33
  5232.1 2064.20  5254.3 2075.18  5267.7 2078.49  5282.2 2079.50  5335.0 2087.02
#Mann=5,-1,0
  4500.6    0.07       0  4635.0    0.16       0  5018.7    0.07       0
  5023.1    0.16       0  5282.2    0.07       0
Bank Sta=5018.7,5023.1
Exp/Cntr=0.3,0.1

Type RM Length L Ch R = 1,2667,139,139,139
BEGIN DESCRIPTION:
Elm 79 2666.91
END DESCRIPTION:
XS GIS Cut Line= 3
      1534495.32      6768285.73      1534675.88      6768716.30
      1534980.72      6768750.95
#Sta/Elev= 30
  4532.3 2065.75  4589.0 2051.17  4595.3 2047.78  4602.2 2047.96  4619.0 2044.35
  4642.8 2041.75  4719.1 2037.16  4748.7 2033.10  4801.7 2031.92  4807.1 2033.63
  4825.5 2034.39  4830.9 2036.38  4849.2 2033.61  4854.7 2031.24  4860.1 2032.04
  4883.9 2028.99  4984.4 2029.92  5001.3 2029.00  5006.2 2025.13  5006.5 2024.63
  5010.6 2025.13  5028.5 2029.57  5159.3 2029.89  5179.5 2031.53  5209.7 2041.07
  5229.8 2051.32  5235.2 2055.36  5260.0 2064.08  5280.1 2070.98  5306.0 2075.96
#Mann=4,-1,0
  4532.3    0.07       0  4602.2    0.16       0  5006.2    0.07       0
  5010.6    0.16       0
Bank Sta=5006.2,5010.6
Exp/Cntr=0.3,0.1

Type RM Length L Ch R = 1,2528,155,155,155
BEGIN DESCRIPTION:
Elm 79 2527.57
END DESCRIPTION:
XS GIS Cut Line= 3
      1534326.88      6768777.07      1534559.56      6768780.54
      1534984.93      6768841.31
#Sta/Elev= 30
  4764.9 2062.69  4803.0 2060.89  4812.9 2062.64  4833.0 2066.79  4853.0 2065.83
  4863.0 2063.41  4903.0 2050.54  4943.0 2031.07  4953.0 2027.09  4963.0 2026.71
  4970.8 2023.87  4971.1 2023.37  4975.3 2023.87  4992.8 2025.45  4997.6 2025.45
  5003.1 2024.03  5011.6 2023.99  5023.3 2026.68  5033.4 2027.54  5255.6 2030.51
  5285.9 2033.55  5294.4 2037.41  5299.5 2035.62  5306.1 2040.17  5336.5 2052.27
  5365.1 2059.94  5370.2 2057.70  5387.0 2061.35  5407.2 2063.10  5427.3 2067.66
#Mann=4,-1,0
  4764.9   0.035       0  4812.9    0.16       0  4970.8    0.07       0
  4975.3    0.16       0
Bank Sta=4970.8,4975.3
Exp/Cntr=0.3,0.1

Type RM Length L Ch R = 1,2373,89,89,89
BEGIN DESCRIPTION:
Elm 79 2372.873
END DESCRIPTION:
XS GIS Cut Line= 3
      1534278.30      6768858.66      1534456.96      6768893.89
      1534967.54      6768898.60
#Sta/Elev= 30
  4817.9 2071.35  4824.7 2067.97  4834.9 2066.15  4865.5 2056.01  4875.7 2055.04
  4885.9 2051.90  4896.6 2044.45  4913.4 2041.42  4916.5 2040.63  4926.7 2034.59
  4942.8 2031.37  4947.9 2027.78  4977.6 2024.52  5008.0 2024.53  5015.8 2022.22
  5016.1 2021.72  5020.3 2022.22  5028.0 2022.43  5038.0 2025.14  5088.0 2024.18
  5168.0 2024.83  5218.0 2027.06  5238.0 2029.01  5298.0 2029.04  5338.1 2030.60
  5368.1 2034.60  5398.1 2040.74  5438.1 2044.00  5468.1 2048.83  5510.6 2053.14
#Mann=4,-1,0
  4817.9    0.07       0  4913.4    0.16       0  5015.8    0.07       0
  5020.3    0.16       0
Bank Sta=5015.8,5020.3
Exp/Cntr=0.3,0.1

Type RM Length L Ch R = 1,2284,80,80,80
BEGIN DESCRIPTION:
Elm 79 3965
END DESCRIPTION:
XS GIS Cut Line= 3
      1534257.48      6768926.37      1534457.36      6768982.10
      1534881.27      6768973.27
#Sta/Elev= 30
  4792.5 2060.64  4810.7 2057.41  4816.5 2052.26  4821.7 2050.51  4831.4 2044.55
  4841.8 2040.09  4850.7 2037.24  4862.6 2032.42  4873.0 2029.87  4883.4 2028.46
  4895.3 2025.10  4909.1 2024.33  4968.8 2024.02  4984.9 2020.98  4985.2 2020.48
  4989.1 2020.48  4989.4 2020.98  5047.6 2023.12  5067.7 2021.87  5087.7 2023.26
  5107.7 2023.41  5127.7 2022.47  5147.7 2023.39  5197.7 2029.13  5277.7 2032.31
  5297.7 2034.66  5317.7 2035.16  5337.7 2038.30  5347.7 2039.25  5424.0 2043.24
#Mann=4,-1,0
  4792.5    0.07       0  4909.1    0.16       0  4984.9    0.07       0
  4989.4    0.16       0
Bank Sta=4984.9,4989.4
Exp/Cntr=0.3,0.1

Type RM Length L Ch R = 1,2204,83,83,83
BEGIN DESCRIPTION:
Elm 79 3963
END DESCRIPTION:
XS GIS Cut Line= 3
      1534184.60      6769002.77      1534493.52      6769047.90
      1534821.73      6769023.72
#Sta/Elev= 30
  4687.8 2047.68  4691.3 2046.16  4738.7 2046.33  4756.2 2045.22  4761.3 2043.20
  4779.2 2041.68  4799.4 2032.48  4809.5 2027.00  4819.6 2024.66  4831.2 2023.13
  4872.9 2023.00  4896.1 2023.16  4901.2 2022.59  4940.9 2023.03  4966.1 2022.40
  4981.3 2021.71  4989.1 2018.79  4989.4 2018.29  4993.3 2018.29  4993.6 2018.79
  4998.2 2020.47  5003.2 2020.47  5011.5 2021.61  5091.7 2022.20  5111.8 2022.89
  5121.8 2024.31  5232.1 2030.75  5262.2 2033.62  5282.2 2036.47  5329.1 2039.16
#Mann=4,-1,0
  4687.8    0.07       0  4872.9    0.16       0  4989.1    0.07       0
  4993.6    0.16       0
Bank Sta=4989.1,4993.6
Exp/Cntr=0.3,0.1

Type RM Length L Ch R = 1,2121,72,72,72
BEGIN DESCRIPTION:
Elm 79 3962
END DESCRIPTION:
XS GIS Cut Line= 3
      1534196.73      6769124.29      1534454.75      6769117.84
      1534807.62      6769082.82
#Sta/Elev= 30
  4741.9 2033.10  4789.3 2033.98  4794.3 2034.78  4820.2 2035.57  4850.2 2035.11
  4860.2 2033.54  4870.2 2027.04  4880.2 2023.09  4890.2 2021.97  4910.4 2022.86
  4920.2 2021.83  4970.2 2021.83  5002.6 2020.87  5010.3 2019.63  5018.1 2019.13
  5018.4 2018.63  5022.3 2018.63  5022.6 2019.13  5030.4 2020.53  5060.5 2020.84
  5080.6 2020.48  5100.7 2021.11  5120.8 2021.14  5148.1 2022.33  5153.1 2022.07
  5161.0 2023.11  5211.3 2025.19  5241.4 2027.21  5281.6 2031.15  5354.6 2036.19
#Mann=5,-1,0
  4741.9   0.035       0  4860.2    0.07       0  4910.4    0.16       0
  5018.1    0.07       0  5022.6    0.16       0
Bank Sta=5018.1,5022.6
Exp/Cntr=0.3,0.1

Type RM Length L Ch R = 1,2049,191,191,191
BEGIN DESCRIPTION:
Elm 79 3961
END DESCRIPTION:
XS GIS Cut Line= 3
      1534021.38      6769254.50      1534454.95      6769190.26
      1534844.25      6769157.28
#Sta/Elev= 30
  4561.7 2039.54  4566.1 2039.54  4571.2 2037.85  4576.2 2037.59  4595.7 2033.42
  4605.8 2030.52  4626.0 2027.17  4705.1 2026.32  4787.8 2028.38  4818.1 2026.92
  4838.3 2027.60  4849.2 2028.76  4858.5 2027.24  4888.9 2019.97  4929.3 2020.21
  4959.6 2018.97  4983.1 2019.16  5017.9 2015.95  5018.2 2015.45  5022.4 2015.95
  5040.2 2018.11  5060.3 2019.23  5110.4 2019.35  5200.1 2021.76  5205.1 2022.82
  5250.9 2025.34  5301.1 2029.93  5324.6 2033.95  5351.3 2037.31  5390.7 2036.84
#Mann=3,-1,0
  4561.7   0.035       0  5017.9   0.035       0  5022.4   0.035       0
Bank Sta=5017.9,5022.4
Exp/Cntr=0.3,0.1

Type RM Length L Ch R = 1,1858,113,113,113
BEGIN DESCRIPTION:
Elm 79 3958
END DESCRIPTION:
XS GIS Cut Line= 3
      1534012.72      6769398.59      1534353.07      6769341.51
      1534769.67      6769273.59
#Sta/Elev= 30
  4654.9 2023.83  4685.6 2023.00  4746.3 2022.67  4778.9 2023.46  4804.3 2021.53
  4806.9 2021.37  4812.0 2022.60  4829.6 2021.64  4872.7 2021.35  4941.1 2018.16
  4959.1 2016.22  4959.4 2015.72  4963.3 2015.72  4963.7 2016.22  4971.5 2016.84
  4994.0 2016.82  4998.4 2017.48  5024.2 2016.90  5111.7 2017.93  5153.9 2017.33
  5204.6 2018.15  5285.7 2017.77  5295.8 2018.24  5301.2 2020.22  5306.2 2020.49
  5326.2 2025.75  5362.6 2028.62  5376.8 2028.16  5407.2 2031.99  5422.1 2032.94
#Mann=5,-1,0
  4654.9    0.07       0  4804.3    0.16       0  4959.1    0.07       0
  4963.7    0.16       0  5024.2   0.035       0
Bank Sta=4959.1,4963.7
Exp/Cntr=0.3,0.1

Type RM Length L Ch R = 1,1745,115,115,115
BEGIN DESCRIPTION:
Elm 79 3960
END DESCRIPTION:
XS GIS Cut Line= 3
      1534003.99      6769419.43      1534300.81      6769436.26
      1534594.28      6769440.26
#Sta/Elev= 30
  4702.7 2024.28  4733.8 2022.76  4743.8 2023.50  4753.8 2022.49  4767.3 2018.60
  4833.9 2018.06  4857.5 2018.49  4884.0 2019.52  4914.1 2018.26  4924.1 2019.13
  4934.1 2018.49  4940.7 2017.20  4945.7 2015.15  4951.8 2014.81  4952.2 2014.31
  4956.1 2014.31  4956.4 2014.81  4956.5 2014.81  5055.5 2016.19  5084.2 2016.23
  5114.2 2017.45  5124.2 2019.02  5154.2 2021.49  5174.2 2021.62  5184.2 2022.37
  5194.2 2024.48  5214.2 2027.44  5234.2 2029.41  5254.2 2030.97  5293.5 2031.48
#Mann=6,-1,0
  4702.7    0.07       0  4857.5    0.16       0  4951.8    0.07       0
  4956.4    0.16       0  4956.5    0.07       0  5055.5    0.16       0
Bank Sta=4951.8,4956.4
Exp/Cntr=0.3,0.1

Type RM Length L Ch R = 1,1630,128,128,128
BEGIN DESCRIPTION:
Elm 79 3959
END DESCRIPTION:
XS GIS Cut Line= 3
      1533972.79      6769435.07      1534250.84      6769536.28
      1534491.79      6769582.28
#Sta/Elev= 30
  4704.1 2025.00  4724.9 2024.47  4738.4 2022.72  4755.4 2021.49  4760.8 2022.09
  4780.7 2020.29  4786.0 2021.92  4802.2 2018.95  4811.3 2018.03  4816.6 2018.60
  4834.2 2017.12  4855.4 2017.01  4872.4 2015.82  4877.8 2016.27  4908.6 2015.18
  4928.3 2015.43  4956.6 2013.46  4956.9 2012.96  4960.8 2012.96  4961.2 2013.46
  5003.7 2013.58  5037.9 2014.85  5084.9 2014.39  5103.9 2017.81  5116.2 2019.45
  5136.6 2023.80  5142.1 2025.64  5156.9 2028.04  5187.5 2029.14  5245.3 2029.07
#Mann=5,-1,0
  4704.1    0.16       0  4956.6    0.07       0  4961.2    0.16       0
  5003.7    0.07       0  5103.9    0.16       0
Bank Sta=4956.6,4961.2
Exp/Cntr=0.3,0.1

Type RM Length L Ch R = 1,1502,102,102,102
BEGIN DESCRIPTION:
Elm 79 3957
END DESCRIPTION:
XS GIS Cut Line= 3
      1533929.97      6769462.98      1534194.37      6769648.00
      1534465.83      6769712.84
#Sta/Elev= 30
  4677.3 2024.75  4727.9 2024.60  4756.7 2026.20  4780.9 2025.16  4793.3 2024.92
  4805.5 2023.11  4831.3 2017.24  4842.1 2015.10  4856.1 2013.49  4864.8 2014.28
  4891.8 2012.69  4958.7 2012.27  4972.0 2012.86  4978.2 2012.13  4993.0 2012.13
  4995.0 2011.53  4995.4 2011.03  4999.6 2011.53  5018.8 2012.71  5042.0 2012.74
  5060.9 2013.85  5066.0 2013.30  5072.6 2016.06  5103.0 2018.64  5108.1 2018.41
  5150.2 2022.87  5159.3 2023.07  5206.3 2026.06  5234.4 2026.71  5279.1 2026.52
#Mann=8,-1,0
  4677.3    0.16       0  4780.9   0.033       0  4831.3    0.16       0
  4958.7    0.07       0  4995.0    0.07       0  4999.6    0.07       0
  5042.0    0.16       0  5159.3   0.035       0
Bank Sta=4995,4999.6
Exp/Cntr=0.3,0.1

Type RM Length L Ch R = 1,1400,68,68,68
BEGIN DESCRIPTION:
Elm 79 3955
END DESCRIPTION:
XS GIS Cut Line= 3
      1533898.14      6769485.44      1534106.46      6769691.90
      1534469.27      6769844.77
#Sta/Elev= 30
  4706.7 2024.44  4713.4 2024.68  4727.5 2023.48  4756.0 2024.34  4798.2 2024.87
  4826.5 2023.64  4840.7 2022.12  4847.7 2019.14  4854.8 2018.58  4861.8 2016.14
  4876.0 2013.92  4899.1 2012.50  4925.7 2011.33  4967.9 2011.58  5017.8 2010.45
  5018.2 2009.95  5022.4 2010.45  5056.2 2011.03  5085.4 2013.01  5097.5 2012.93
  5117.8 2012.77  5127.4 2013.55  5132.8 2012.95  5156.6 2014.24  5162.0 2013.77
  5180.3 2015.65  5260.2 2019.05  5356.5 2025.08  5368.1 2026.76  5393.7 2026.24
#Mann=8,-1,0
  4706.7    0.16       0  4756.0   0.033       0  4899.1    0.16       0
  4925.7    0.07       0  5017.8    0.07       0  5022.4    0.07       0
  5097.5    0.16       0  5260.2   0.035       0
Bank Sta=5017.8,5022.4
Exp/Cntr=0.3,0.1

Type RM Length L Ch R = 1,1332,109,109,109
BEGIN DESCRIPTION:
Elm 79 3954
END DESCRIPTION:
XS GIS Cut Line= 3
      1533846.85      6769550.35      1534058.89      6769739.43
      1534430.01      6769913.00
#Sta/Elev= 30
  4715.9 2022.58  4720.0 2021.97  4762.6 2022.94  4791.1 2022.26  4805.3 2019.58
  4819.5 2018.28  4826.2 2016.52  4833.7 2016.85  4840.4 2014.97  4860.1 2013.17
  4903.9 2011.18  4969.1 2010.86  5004.8 2010.99  5025.4 2009.77  5025.7 2009.27
  5030.0 2009.77  5061.9 2011.54  5073.0 2011.08  5101.7 2012.02  5116.5 2011.20
  5130.1 2010.85  5195.6 2012.74  5205.8 2013.28  5238.6 2014.32  5267.1 2017.02
  5295.5 2018.43  5326.9 2021.60  5381.3 2025.07  5391.1 2024.81  5409.7 2024.24
#Mann=9,-1,0
  4715.9   0.033       0  4860.1    0.16       0  4969.1    0.07       0
  5025.4    0.07       0  5030.0    0.07       0  5116.5    0.16       0
  5195.6    0.12       0  5205.8   0.035       0  5391.1    0.07       0
Bank Sta=5025.4,5030
Exp/Cntr=0.3,0.1

Type RM Length L Ch R = 1,1223,144,144,144
BEGIN DESCRIPTION:
Elm 79 3953
END DESCRIPTION:
XS GIS Cut Line= 3
      1533813.05      6769669.44      1534010.17      6769831.84
      1534406.77      6769999.29
#Sta/Elev= 30
  4744.6 2020.52  4766.2 2020.70  4787.1 2018.62  4794.9 2016.15  4801.4 2015.61
  4809.3 2013.83  4815.1 2013.80  4858.8 2011.06  4922.9 2009.67  4972.1 2010.59
  4980.0 2009.85  4986.5 2010.27  4991.0 2009.13  4991.3 2008.63  4995.6 2009.13
  5025.1 2010.55  5054.2 2010.92  5063.1 2010.38  5136.2 2009.16  5183.6 2009.43
  5212.8 2010.42  5225.9 2012.02  5236.5 2012.36  5265.8 2017.35  5289.3 2020.44
  5313.0 2021.69  5365.9 2022.29  5385.8 2023.47  5418.7 2022.58  5430.5 2023.11
#Mann=8,-1,0
  4744.6   0.033       0  4815.1    0.16       0  4922.9    0.07       0
  4991.0    0.07       0  4995.6    0.07       0  5063.1    0.12       0
  5225.9   0.035       0  5385.8    0.07       0
Bank Sta=4991,4995.6
Exp/Cntr=0.3,0.1

Type RM Length L Ch R = 1,1079,97,97,97
BEGIN DESCRIPTION:
Elm 79 3952
END DESCRIPTION:
XS GIS Cut Line= 3
      1533797.43      6769792.72      1533910.52      6769935.57
      1534306.06      6770077.40
#Sta/Elev= 30
  4817.8 2020.34  4848.9 2019.75  4898.6 2014.88  4901.8 2013.94  4905.0 2012.99
  4919.4 2011.28  4940.2 2009.58  4968.4 2008.96  5015.4 2008.39  5021.3 2008.85
  5052.1 2009.16  5068.5 2008.65  5077.5 2008.99  5082.8 2008.44  5121.6 2007.65
  5214.9 2007.45  5215.2 2006.95  5219.2 2006.95  5219.5 2007.45  5262.0 2008.25
  5291.8 2010.43  5312.8 2012.15  5318.2 2013.29  5343.6 2015.25  5355.3 2016.70
  5366.0 2016.88  5374.4 2018.43  5387.2 2019.56  5410.5 2021.25  5420.2 2021.15
#Mann=6,-1,0
  4817.8   0.033       0  4901.8    0.16       0  4968.4    0.12       0
  5214.9    0.07       0  5219.5    0.12       0  5291.8   0.035       0
Bank Sta=5214.9,5219.5
Exp/Cntr=0.3,0.1

Type RM Length L Ch R = 1,982,82,82,82
BEGIN DESCRIPTION:
Elm 79 3951
END DESCRIPTION:
XS GIS Cut Line= 3
      1533780.24      6769889.46      1533902.64      6770032.02
      1534186.11      6770139.06
#Sta/Elev= 30
  4812.1 2019.40  4836.8 2018.89  4849.7 2017.01  4857.0 2016.39  4871.3 2013.64
  4885.6 2012.51  4892.2 2011.49  4899.8 2011.13  4913.8 2009.41  4928.4 2008.59
  4969.0 2008.50  4984.4 2007.98  4998.0 2008.57  5005.3 2008.13  5023.9 2008.80
  5045.3 2007.86  5077.3 2007.74  5098.7 2007.05  5148.0 2006.87  5173.5 2006.67
  5173.8 2006.17  5177.8 2006.17  5178.1 2006.67  5216.3 2007.39  5248.4 2008.65
  5272.9 2010.71  5280.4 2011.34  5285.8 2012.37  5291.2 2012.07  5303.0 2012.98
#Mann=8,-1,0
  4812.1   0.033       0  4836.8    0.16       0  4913.8    0.12       0
  4969.0   0.033       0  5148.0    0.12       0  5173.5   0.033       0
  5178.1    0.12       0  5272.9   0.035       0
Bank Sta=5173.5,5178.1
Exp/Cntr=0.3,0.1

Type RM Length L Ch R = 1,900,67,67,67
BEGIN DESCRIPTION:
Elm 79 3950
END DESCRIPTION:
XS GIS Cut Line= 3
      1533760.72      6769930.68      1533856.23      6770098.51
      1534133.99      6770215.00
#Sta/Elev= 30
  4806.9 2018.59  4823.4 2017.69  4838.3 2015.53  4866.6 2012.67  4882.5 2012.14
  4888.2 2010.14  4895.9 2009.50  4918.9 2008.71  4925.7 2009.00  4931.4 2008.48
  4953.4 2008.56  4974.1 2007.89  5013.3 2006.61  5031.2 2007.89  5084.6 2006.92
  5096.3 2007.29  5107.1 2006.59  5128.8 2006.83  5159.0 2005.89  5159.3 2005.39
  5163.3 2005.39  5163.6 2005.89  5183.0 2006.53  5190.5 2007.22  5197.8 2006.86
  5219.7 2008.03  5231.5 2009.37  5237.2 2009.68  5272.7 2013.89  5301.2 2015.85
#Mann=6,-1,0
  4806.9    0.16       0  4974.1   0.033       0  5159.0   0.033       0
  5163.6   0.033       0  5197.8    0.12       0  5231.5   0.035       0
Bank Sta=5159,5163.6
Exp/Cntr=0.3,0.1

Type RM Length L Ch R = 1,833,140,140,140
BEGIN DESCRIPTION:
Elm 79 3949
END DESCRIPTION:
XS GIS Cut Line= 3
      1533725.99      6770017.49      1533854.55      6770165.31
      1534097.84      6770253.54
#Sta/Elev= 30
  4804.1 2015.89  4831.7 2014.56  4867.8 2010.62  4882.0 2009.68  4919.1 2008.10
  4931.4 2007.30  4952.3 2006.88  4966.5 2006.10  4988.4 2005.92  5019.5 2006.77
  5024.8 2006.11  5050.1 2006.69  5055.4 2005.46  5074.9 2005.66  5083.8 2005.19
  5084.1 2004.69  5088.1 2004.69  5088.4 2005.19  5117.5 2005.51  5149.4 2005.20
  5181.3 2006.53  5194.1 2007.93  5197.9 2008.75  5203.2 2008.80  5213.2 2010.32
  5223.2 2013.31  5228.5 2014.04  5234.5 2014.56  5245.1 2014.71  5258.8 2015.95
#Mann=5,-1,0
  4804.1    0.16       0  4919.1   0.033       0  5083.8   0.033       0
  5088.4   0.033       0  5194.1   0.035       0
Bank Sta=5083.8,5088.4
Exp/Cntr=0.3,0.1

Type RM Length L Ch R = 1,693,140,140,140
BEGIN DESCRIPTION:
Elm 79 3948
END DESCRIPTION:
XS GIS Cut Line= 3
      1533730.00      6770106.49      1533808.65      6770289.51
      1534077.53      6770286.62
#Sta/Elev= 30
  4800.8 2009.23  4822.4 2008.41  4846.0 2007.12  4851.4 2006.59  4875.0 2005.65
  4898.5 2005.20  4927.5 2005.13  4943.9 2004.43  4951.1 2004.47  4956.5 2004.14
  4980.1 2004.05  5004.1 2003.28  5004.4 2002.78  5008.4 2002.78  5008.7 2003.28
  5036.4 2003.47  5066.4 2004.30  5076.4 2004.38  5096.4 2004.46  5106.4 2004.26
  5116.4 2004.43  5126.4 2004.19  5166.4 2004.41  5186.4 2005.33  5206.4 2006.97
  5216.4 2008.13  5226.8 2010.10  5246.4 2014.17  5265.2 2015.91  5268.9 2015.91
#Mann=4,-1,0
  4800.8   0.033       0  5004.1   0.033       0  5008.7   0.033       0
  5226.8   0.035       0
Bank Sta=5004.1,5008.7
Exp/Cntr=0.3,0.1

Type RM Length L Ch R = 1,553,91,91,91
BEGIN DESCRIPTION:
Elm 79 3947
END DESCRIPTION:
XS GIS Cut Line= 3
      1533561.05      6770405.97      1533869.62      6770402.04
      1534029.97      6770338.71
#Sta/Elev= 30
  4691.4 2005.09  4715.4 2005.02  4775.4 2004.09  4785.4 2003.73  4825.4 2004.00
  4835.4 2003.64  4845.4 2003.64  4875.4 2003.96  4915.4 2003.58  4935.4 2003.10
  4945.4 2003.34  5000.0 2003.29  5003.3 2003.04  5003.7 2002.54  5007.9 2002.54
  5008.2 2003.04  5023.3 2003.19  5028.6 2003.56  5047.6 2003.54  5059.5 2003.84
  5070.3 2004.31  5077.4 2005.01  5091.8 2005.30  5101.7 2005.97  5107.1 2006.06
  5136.8 2008.04  5155.8 2010.33  5161.2 2010.68  5167.1 2013.06  5172.4 2013.91
#Mann=3,-1,0
  4691.4   0.033       0  5003.3   0.033       0  5008.2   0.033       0
Bank Sta=5003.3,5008.2
Exp/Cntr=0.3,0.1

Type RM Length L Ch R = 1,462,132,132,132
BEGIN DESCRIPTION:
Elm 79 3946
END DESCRIPTION:
XS GIS Cut Line= 3
      1533729.98      6770563.01      1533934.25      6770466.08
      1534030.01      6770362.99
#Sta/Elev= 30
  4773.9 2003.78  4790.5 2003.89  4796.7 2003.57  4812.7 2003.72  4819.4 2003.49
  4847.7 2003.15  4864.9 2003.24  4879.1 2003.07  4887.6 2003.29  4893.1 2003.06
  4910.3 2002.89  4915.8 2003.04  4967.6 2002.87  4976.1 2002.51  4976.4 2002.01
  4980.6 2002.01  4981.0 2002.51  4989.8 2002.66  5002.1 2002.54  5020.5 2003.03
  5041.5 2003.03  5048.8 2003.71  5055.7 2003.72  5063.0 2004.00  5069.8 2004.74
  5084.0 2005.47  5091.4 2006.18  5119.7 2008.08  5126.5 2008.66  5140.7 2010.42
#Mann=3,-1,0
  4773.9   0.033       0  4976.1   0.033       0  4981.0   0.033       0
Bank Sta=4976.1,4981
Exp/Cntr=0.3,0.1

Type RM Length L Ch R = 1,330,213,213,213
BEGIN DESCRIPTION:
Elm 79 3945
END DESCRIPTION:
XS GIS Cut Line= 3
      1533890.90      6770644.72      1534038.68      6770537.63
      1534179.57      6770349.55
#Sta/Elev= 30
  4817.5 2002.52  4839.3 2002.69  4847.3 2002.41  4896.7 2002.41  4910.4 2002.66
  4918.9 2002.30  4969.2 2002.17  4990.1 2001.97  5001.5 2001.59  5001.9 2001.09
  5006.1 2001.09  5006.4 2001.59  5018.6 2002.06  5024.8 2001.74  5042.9 2002.27
  5047.8 2002.44  5054.0 2003.44  5068.6 2004.56  5074.8 2005.30  5083.2 2004.94
  5089.4 2005.41  5124.8 2008.98  5139.4 2010.22  5154.0 2011.95  5162.0 2012.40
  5168.6 2013.27  5183.2 2014.41  5189.4 2013.66  5204.0 2015.54  5235.0 2015.72
#Mann=4,-1,0
  4817.5   0.033       0  5001.5   0.033       0  5006.4   0.033       0
  5042.9   0.035       0
Bank Sta=5001.5,5006.4
Exp/Cntr=0.3,0.1

Type RM Length L Ch R = 1,117,0,0,0
BEGIN DESCRIPTION:
Elm 79 3944
END DESCRIPTION:
XS GIS Cut Line= 3
      1533895.31      6770670.73      1534206.64      6770633.97
      1534289.62      6770442.15
#Sta/Elev= 30
  4686.5 2002.42  4746.6 2001.68  4757.1 2002.05  4776.8 2001.89  4786.9 2001.51
  4797.0 2001.77  4817.1 2001.46  4840.0 2001.46  4847.3 2001.70  4922.9 2000.62
  4927.9 2000.96  4958.1 2001.14  4985.8 1999.94  4986.2 1999.44  4990.4 1999.44
  4990.8 1999.94  5017.4 1999.96  5062.6 2002.64  5071.9 2003.83  5086.1 2004.50
  5109.6 2006.53  5115.5 2007.60  5126.4 2008.71  5136.5 2010.26  5156.6 2013.30
  5162.0 2012.82  5180.1 2013.66  5191.7 2013.21  5202.6 2013.76  5209.0 2013.72
#Mann=4,-1,0
  4686.5   0.033       0  4985.8   0.033       0  4990.8   0.033       0
  5136.5   0.035       0
Bank Sta=4985.8,4990.8
Exp/Cntr=0.3,0.1

Chan Stop Cuts=-1
