HEC-RAS study Elm 85.prj: Elm 85 Base Level Engineering

--- Elm 85.g01 (geometry) --- (continued)

Type RM Length L Ch R = 1 ,23599   ,102,102,102
BEGIN DESCRIPTION:
692
END DESCRIPTION:
XS GIS Cut Line= 3
      1530117.56      6789959.42      1529848.43      6789672.93
      1529349.63       6789529.8
#Sta/Elev= 30
  4584.1 2201.13  4737.2 2194.57  4855.8 2190.16    4870 2187.13  4876.8 2182.59
  4884.1 2182.25    4891 2176.76  4933.5 2169.99    4955    2170  4969.1 2166.09
    4976 2157.14  4991.1 2150.47  4997.5 2150.02    4998 2149.52  5005.5 2150.02
    5010 2154.79  5015.2 2154.49  5022.4 2160.74  5032.8 2162.49  5048.9 2171.11
  5054.1 2168.75  5074.4 2172.99  5160.5 2174.01  5188.8  2178.5  5240.8 2194.15
  5266.9 2197.76  5272.1 2200.44  5292.8 2199.05  5386.5  2205.4  5496.1 2207.77
#Mann= 4 ,-1 , 0
  4584.1     .07       0  4737.2     .16       0  4997.5     .07       0
  5005.5     .16       0
Bank Sta=4997.5,5005.5
XS Rating Curve= 0 ,0
Exp/Cntr=0.3,0.1

Type RM Length L Ch R = 1 ,23497   ,91,91,91
BEGIN DESCRIPTION:
693
END DESCRIPTION:
XS GIS Cut Line= 3
      1530239.09      6789777.12      1529852.77       6789573.1
      1529362.36        6789508.
#Sta/Elev= 30
  4564.6 2209.28  4590.5 2208.38  4656.6 2196.37  4710.8 2191.53    4827 2187.09
  4863.3 2184.27  4885.9  2180.2  4898.7  2182.6  4931.1 2183.32  4937.1 2180.02
  4942.8  2180.2  4959.1 2174.24    4965 2169.84  4975.5 2165.41  4981.1 2166.74
  4987.7 2158.93  4997.4 2150.98  5005.3 2149.34  5005.8 2148.84  5013.3 2149.34
  5019.4 2152.48  5029.5 2154.17  5039.6 2159.43  5059.8 2163.63  5076.6 2170.54
  5154.9 2174.94  5180.8 2185.65  5228.2 2196.96  5392.7 2205.41  5496.2  2208.6
#Mann= 4 ,-1 , 0
  4564.6     .07       0  4710.8     .16       0  5005.3     .07       0
  5013.3     .16       0
Bank Sta=5005.3,5013.3
XS Rating Curve= 0 ,0
Exp/Cntr=0.3,0.1

Type RM Length L Ch R = 1 ,23406   ,156,156,156
BEGIN DESCRIPTION:
691
END DESCRIPTION:
XS GIS Cut Line= 3
      1530282.46      6789716.34      1529844.09      6789477.62
      1529319.42      6789486.29
#Sta/Elev= 30
  4512.8  2204.2  4523.4 2207.43  4561.4 2208.87  4583.2 2205.92  4589.6 2202.77
  4612.4 2196.85  4659.5 2192.02  4730.4 2186.22  4850.1 2186.73  4871.9 2185.49
  4885.7 2183.17  4921.3 2172.58  4943.1 2170.84  4959.3 2166.41  4965.4 2159.53
  4975.4 2152.33  4993.3 2148.35  4993.8 2147.85  5001.3 2148.35  5008.6  2153.2
    5014  2153.2    5021 2159.05  5041.1 2167.66  5101.1 2171.81  5161.1 2195.47
  5171.1  2196.9  5191.1 2197.95  5211.1 2196.68  5231.1 2199.22  5536.7 2210.05
#Mann= 4 ,-1 , 0
  4512.8     .07       0  4659.5     .16       0  4993.3     .07       0
  5001.3     .16       0
Bank Sta=4993.3,5001.3
XS Rating Curve= 0 ,0
Exp/Cntr=0.3,0.1

Type RM Length L Ch R = 1 ,23250   ,142,142,142
BEGIN DESCRIPTION:
690
END DESCRIPTION:
XS GIS Cut Line= 3
      1530282.42       6789672.9      1529943.91      6789360.43
      1529392.74      6789195.51
#Sta/Elev= 30
  4530.3 2204.44  4581.2 2203.05  4669.9 2189.79    4829 2176.96  4836.4 2179.33
  4857.4 2177.83  4885.7  2172.4  4893.1 2174.62  4907.3 2173.53  4949.2 2162.69
  4963.4 2161.28  4984.9 2151.95  5010.7 2149.63  5012.4 2146.01  5012.9 2145.51
  5020.4 2146.01  5031.6 2155.18  5087.8 2161.61  5104.7 2170.28  5115.1 2172.89
  5192.4 2174.38  5263.8 2180.64  5291.7 2188.79  5296.9 2187.65  5313.4 2195.06
  5335.2 2193.42  5376.1 2200.01  5472.8 2204.06  5511.8 2199.87  5566.3 2200.68
#Mann= 4 ,-1 , 0
  4530.3     .07       0  4669.9     .16       0  5012.4     .07       0
  5020.4     .16       0
Bank Sta=5012.4,5020.4
XS Rating Curve= 0 ,0
Exp/Cntr=0.3,0.1

Type RM Length L Ch R = 1 ,23108   ,88,88,88
BEGIN DESCRIPTION:
688
END DESCRIPTION:
XS GIS Cut Line= 3
      1530338.85      6789525.34      1530004.68       6789238.9
      1529653.15      6788974.17
#Sta/Elev= 30
  4565.5 2184.13  4580.8 2189.32  4587.4 2187.79  4595.1  2191.4  4601.7 2188.66
  4609.3 2191.23  4615.9 2188.75  4630.2 2192.83  4636.8 2190.33  4717.1 2188.04
  4892.5 2186.34  4913.4 2178.75  4963.9 2153.88  4998.4  2144.2  4998.9  2143.7
  5006.5  2144.2  5019.7 2151.41  5034.3 2152.71  5055.3 2162.61  5063.4 2162.16
  5069.7 2165.36    5078 2162.09  5084.3  2164.1  5092.6 2161.05  5098.8 2163.53
  5148.8 2167.13  5163.4 2171.26  5384.1 2178.31  5427.8 2181.29  5445.7 2185.33
#Mann= 4 ,-1 , 0
  4565.5     .07       0  4717.1     .16       0  4998.4     .07       0
  5006.5     .16       0
Bank Sta=4998.4,5006.5
XS Rating Curve= 0 ,0
Exp/Cntr=0.3,0.1

Type RM Length L Ch R = 1 ,23020   ,161,161,161
BEGIN DESCRIPTION:
689
END DESCRIPTION:
XS GIS Cut Line= 3
      1530330.21      6789468.94      1530074.12      6789182.48
      1529705.16      6788909.01
#Sta/Elev= 30
  4606.5 2179.83  4653.3 2189.67  4753.4 2186.52  4830.8 2186.39  4897.4 2184.39
  4949.8 2172.62  4997.2 2144.52  4997.7 2144.02  5005.3 2144.52  5036.7 2153.14
    5043 2158.67  5057.6 2165.53  5086.8 2165.42  5107.7 2158.58  5157.7 2164.76
    5164    2162  5193.2 2161.03  5207.8 2165.06  5214.1 2163.53  5237.1 2167.74
  5243.3 2166.42  5257.9 2170.55  5272.5 2168.58  5278.8 2164.21  5300.8 2171.17
  5372.7 2176.91  5393.6 2184.99  5422.8 2190.71    5429 2194.98    5450 2195.78
#Mann= 6 ,-1 , 0
  4606.5     .07       0  4753.4     .16       0  4830.8     .07       0
  4897.4     .16       0  4997.2     .07       0  5005.3     .16       0
Bank Sta=4997.2,5005.3
XS Rating Curve= 0 ,0
Exp/Cntr=0.3,0.1

Type RM Length L Ch R = 1 ,22859   ,108,108,108
BEGIN DESCRIPTION:
686
END DESCRIPTION:
XS GIS Cut Line= 3
      1530360.56      6789464.56      1530156.59      6789047.93
      1529728.43      6788848.99
#Sta/Elev= 30
  4538.8 2179.02  4590.9 2186.54  4607.8 2184.44    4717 2183.47    4821 2182.51
  4827.6 2182.39  4900.4 2182.94  4913.5 2180.59  4945.4 2162.34  4967.9 2154.28
  4980.3 2145.23  4991.9 2141.65  4992.4 2141.15  5000.1 2141.65  5040.6 2157.98
  5057.9 2159.59  5063.5 2162.75  5103.7 2162.17  5114.8 2168.73  5137.6 2175.35
  5223.7 2171.53    5258 2174.73  5303.4 2177.18  5343.7 2189.19  5366.6 2193.14
  5389.5 2192.59    5395 2187.16  5412.4 2189.06  5417.9 2186.01  5474.8 2190.56
#Mann= 7 ,-1 , 0
  4538.8     .07       0    4717     .16       0    4821     .07       0
  4827.6     .16       0  4991.9     .07       0  5000.1     .16       0
    5258    .035       0
Bank Sta=4991.9,5000.1
XS Rating Curve= 0 ,0
Exp/Cntr=0.3,0.1

Type RM Length L Ch R = 1 ,22751   ,189,189,189
BEGIN DESCRIPTION:
687
END DESCRIPTION:
XS GIS Cut Line= 3
      1530555.87      6789356.06      1530247.73      6789000.18
      1529992.77      6788641.51
#Sta/Elev= 30
  4523.7 2197.48  4558.7 2194.66  4600.5  2175.7  4657.5 2162.52  4693.1 2158.55
  4709.4 2162.93  4728.7 2173.41  4778.1 2173.18  4820.8 2162.44  4841.7 2169.73
  4877.8 2167.36  4884.5  2172.3  4927.2 2162.94  4933.8 2166.86  4962.3 2167.09
  4990.8  2150.3  5012.3 2143.59    5016 2141.87  5016.5 2141.37  5024.6 2141.87
  5076.8 2153.23  5112.5 2153.83  5127.3 2166.19  5133.4 2163.53    5142 2168.73
  5198.6 2175.17  5213.4 2182.45    5240 2182.98  5291.6 2191.22  5434.5 2192.55
#Mann= 6 ,-1 , 0
  4523.7     .07       0  4709.4     .16       0  5012.3    .035       0
    5016     .07       0  5024.6    .035       0    5240     .07       0
#XS Ineff= 2 , 0
       0    5010    2160    5030       0    2160
Permanent Ineff=
       F       F
Bank Sta=5016,5024.6
XS Rating Curve= 0 ,0
Exp/Cntr=0.3,0.1

Type RM Length L Ch R = 1 ,22562   ,139,139,139
BEGIN DESCRIPTION:
684
END DESCRIPTION:
XS GIS Cut Line= 3
      1530798.97      6789160.79       1530351.9      6788848.27
      1530009.49      6788549.21
#Sta/Elev= 30
  4449.8 2204.03    4519 2199.33    4529 2197.79  4576.7 2193.58  4696.9 2177.62
  4874.8 2158.74  4881.9 2157.87  4935.6 2150.49  4956.6 2140.21  4967.1 2138.44
  4967.6 2137.94  4975.7 2138.44  4991.1 2146.69  5003.3 2146.28  5014.8 2148.01
    5029 2154.36  5035.7 2160.08  5043.3 2160.36  5047.1 2164.65  5049.9 2167.81
  5057.5 2166.81  5064.1 2169.58  5078.4 2167.88  5156.2 2176.25  5184.7 2186.61
  5198.9 2188.64  5311.9 2189.93  5326.1 2193.29    5348 2191.09  5449.9 2191.71
#Mann= 10 ,-1 , 0
  4449.8     .07       0    4519    .035       0    4529     .07       0
  4696.9    .035       0  4874.8     .07       0  4881.9     .16       0
  4967.1     .07       0  4975.7     .16       0  5003.3    .035       0
  5047.1     .07       0
Bank Sta=4967.1,4975.7
XS Rating Curve= 0 ,0
Exp/Cntr=0.3,0.1

Type RM Length L Ch R = 1 ,22423   ,149,149,149
BEGIN DESCRIPTION:
685
END DESCRIPTION:
XS GIS Cut Line= 3
      1530881.39      6789056.59      1530430.02      6788735.43
      1530058.39      6788497.76
#Sta/Elev= 30
  4466.2 2205.22  4519.3 2203.76  4641.5 2195.51    4678 2192.47  4684.1 2193.89
    4695 2189.96  4698.9  2190.2  4713.6 2183.42  4778.8 2169.72  4814.5  2163.7
  4855.6 2160.22    4871 2158.29  4885.8 2159.59  4906.7 2154.75  4915.3 2154.91
  4921.4 2151.72    4951 2146.14  4973.7 2136.24  4974.2 2135.74  4982.3 2136.24
  4992.8 2143.97  5020.2 2146.61  5022.4 2150.68  5049.9 2167.41    5060 2170.39
  5239.8  2175.6  5267.7 2178.79  5298.1 2186.48  5325.2 2188.68  5461.3 2190.63
#Mann= 8 ,-1 , 0
  4466.2    .035       0  4519.3     .07       0  4641.5    .035       0
    4695     .07       0  4855.6     .16       0  4973.7     .07       0
  4982.3     .16       0    5060     .07       0
Bank Sta=4973.7,4982.3
XS Rating Curve= 0 ,0
Exp/Cntr=0.3,0.1

Type RM Length L Ch R = 1 ,22274   ,147,147,147
BEGIN DESCRIPTION:
683
END DESCRIPTION:
XS GIS Cut Line= 3
      1530885.73       6788939.4      1530560.23      6788644.28
       1530004.7      6788383.88
#Sta/Elev= 30
  4548.6 2204.31  4663.3 2200.85  4705.9 2195.33  4755.2 2192.61  4770.2 2189.68
    4812 2172.96  4840.4 2164.63  4903.9 2157.15  4932.3 2150.93  4939.7 2147.97
    4988 2143.95  4995.1 2141.91  5004.8 2135.41  5013.6 2134.65  5014.1 2134.15
  5022.2 2134.65  5026.9 2141.29    5049 2150.99  5058.1 2153.01  5063.6 2156.07
  5080.9 2153.92  5093.1 2160.91  5104.7  2163.6  5115.2 2165.61  5177.7 2169.64
  5297.4  2172.3  5325.7 2175.94    5343 2180.38  5388.7 2188.37  5601.5 2189.88
#Mann= 5 ,-1 , 0
  4548.6     .07       0  4770.2     .16       0  5013.6     .07       0
  5022.2     .16       0  5104.7     .07       0
Bank Sta=5013.6,5022.2
XS Rating Curve= 0 ,0
Exp/Cntr=0.3,0.1

Type RM Length L Ch R = 1 ,22127   ,267,267,267
BEGIN DESCRIPTION:
682
END DESCRIPTION:
XS GIS Cut Line= 3
      1530933.47      6788817.87       1530599.3      6788509.73
      1530243.41      6788314.43
#Sta/Elev= 30
  4532.8 2201.36  4708.3 2198.21  4750.8 2192.89  4767.5  2186.6  4793.4 2178.09
  4800.7  2172.7  4850.1 2162.79  4892.6 2147.86  4984.5 2141.89  4986.9 2136.92
  5010.8  2133.7  5011.3  2133.2  5019.4  2133.7  5049.3 2155.83  5081.1 2169.06
  5086.9  2167.4  5130.5 2178.62  5146.5 2174.84  5168.3 2179.28  5184.4  2175.2
  5190.1 2178.68  5206.2 2176.42  5215.1 2178.92    5228 2177.56  5233.7 2181.75
  5249.8 2180.67  5255.5  2183.5  5287.7 2182.15  5331.3 2188.06  5393.3 2188.83
#Mann= 5 ,-1 , 0
  4532.8     .07       0  4767.5     .16       0  5010.8     .07       0
  5019.4     .16       0  5215.1     .07       0
Bank Sta=5010.8,5019.4
XS Rating Curve= 0 ,0
Exp/Cntr=0.3,0.1

Type RM Length L Ch R = 1 ,21860   ,228,228,228
BEGIN DESCRIPTION:
681
END DESCRIPTION:
XS GIS Cut Line= 4
       1530825.4      6788110.52      1530568.43      6788254.63
      1530420.86      6788348.38      1530160.96      6788266.69
#Sta/Elev= 30
  4708.1 2183.39    4743 2180.64  4751.4 2181.32  4757.1 2179.68  4794.8 2181.58
  4859.8 2161.11  4891.7 2156.17  4912.4 2155.55  4940.8 2153.37  4962.5 2149.34
  4978.5 2143.86  4984.2 2143.75  4994.4 2140.81  5002.7  2131.2  5011.2 2130.81
  5011.7 2130.31  5019.9 2130.81  5030.5 2132.02  5042.6 2138.23  5073.1 2140.34
    5079 2142.14  5094.3 2149.74  5115.5 2163.99  5137.1 2174.66  5160.8 2183.84
  5172.5 2186.04  5194.5 2185.83    5257 2185.83  5340.9 2188.49    5450 2188.16
#Mann= 5 ,-1 , 0
  4708.1     .07       0  4912.4     .16       0  5011.2     .07       0
  5019.9     .16       0  5194.5     .07       0
Bank Sta=5011.2,5019.9
XS Rating Curve= 0 ,0
Exp/Cntr=0.3,0.1

Type RM Length L Ch R = 1 ,21632   ,281,281,281
BEGIN DESCRIPTION:
680
END DESCRIPTION:
XS GIS Cut Line= 3
      1530963.84      6788088.72      1530456.07      6788071.37
      1530088.57      6788084.34
#Sta/Elev= 30
  4490.3 2187.69  4539.2 2185.73  4559.2 2186.63  4639.2 2183.19  4669.2 2184.75
  4719.3 2183.56  4739.3 2177.95  4789.3 2158.45  4809.3 2153.43  4857.5 2145.45
  4899.4 2138.56  4952.5 2135.99  4959.4 2131.92  4975.1 2127.17  4975.6 2126.67
  4983.8 2127.17  4989.4 2128.79  4996.4 2135.43  5001.4 2135.43  5044.6 2144.55
  5049.6 2142.57  5059.5 2144.52  5081.1 2152.18  5119.5 2168.46  5129.5 2174.58
  5139.5  2183.2  5149.5 2184.21  5269.6 2184.21  5326.4 2180.09  5366.1 2179.46
#Mann= 5 ,-1 , 0
  4490.3     .07       0  4857.5     .16       0  4975.1     .07       0
  4983.8     .16       0  5081.1     .07       0
Bank Sta=4975.1,4983.8
XS Rating Curve= 0 ,0
Exp/Cntr=0.3,0.1

Type RM Length L Ch R = 1 ,21351   ,292,292,292
BEGIN DESCRIPTION:
679
END DESCRIPTION:
XS GIS Cut Line= 3
       1531076.7      6787902.09      1530547.21      6787819.63
      1530109.46      6787880.31
#Sta/Elev= 30
    4471 2188.83    4505 2188.78    4603 2187.27  4785.7 2181.76  4847.2  2175.4
  4853.6 2171.74  4858.7 2171.36  4881.5 2163.93  4921.5 2154.44  4938.3 2144.89
  4985.1 2123.72  4985.6 2123.22  4993.8 2123.72    4999 2124.54  5005.5 2128.39
  5010.5 2128.39  5019.2 2132.41  5059.6 2143.05  5089.9 2159.31    5099 2162.89
  5110.1 2167.38  5120.2  2169.2  5150.4 2171.86  5176.4  2169.7  5181.4 2171.83
  5231.2 2162.43  5281.7 2163.84  5372.5 2170.46  5391.6 2173.96  5448.8 2180.75
#Mann= 7 ,-1 , 0
    4471     .07       0    4505     .16       0    4603     .07       0
  4881.5     .16       0  4985.1     .07       0  4993.8     .16       0
    5099     .07       0
Bank Sta=4985.1,4993.8
XS Rating Curve= 0 ,0
Exp/Cntr=0.3,0.1

Type RM Length L Ch R = 1 ,21059   ,215,215,215
BEGIN DESCRIPTION:
678
END DESCRIPTION:
XS GIS Cut Line= 3
      1530994.26        6787633.      1530555.89      6787528.83
       1530169.8      6787641.62
#Sta/Elev= 30
  4548.5 2184.19  4667.8 2183.54  4741.8 2182.78  4784.1 2178.53  4845.8 2156.15
  4851.1 2152.77    4928 2139.82  4958.9 2129.31  4973.3 2119.39  4973.8 2118.89
    4982 2119.39  4989.7 2120.83    4997 2125.79  5002.1 2125.79  5009.6 2130.61
  5014.8 2129.69  5048.2 2153.11  5086.9 2153.26  5114.6 2150.23  5120.4 2147.19
  5185.2 2150.71  5218.8 2154.04    5250 2162.54  5291.7  2168.7  5303.3 2172.72
    5323 2174.14  5336.7 2174.76  5343.8 2169.39  5370.2 2160.51  5401.3 2160.71
#Mann= 6 ,-1 , 0
  4548.5     .16       0  4667.8     .07       0  4741.8     .16       0
  4973.3     .07       0    4982     .16       0  5185.2     .07       0
Bank Sta=4973.3,4982
XS Rating Curve= 0 ,0
Exp/Cntr=0.3,0.1

Type RM Length L Ch R = 1 ,20844   ,249,249,249
BEGIN DESCRIPTION:
677
END DESCRIPTION:
XS GIS Cut Line= 3
      1530855.33      6787437.66      1530594.96      6787324.84
      1530130.53      6787376.92
#Sta/Elev= 30
  4726.8 2180.94  4799.7 2177.55  4816.9  2173.5  4834.9 2177.86  4840.4  2176.5
    4847  2174.4  4857.9 2167.97  4863.8 2162.55  4879.7 2155.76  4887.3 2150.31
  4901.5  2145.1  4934.2 2137.76  4939.7 2134.72  4963.2 2130.23  4986.7 2129.97
  4992.1 2127.49  5003.4 2117.66  5003.9 2117.16  5012.2 2117.66  5020.6 2117.84
  5040.7 2130.04  5060.8 2129.78  5079.9 2135.29  5084.9 2132.19  5101.1 2132.65
  5141.3 2136.43  5161.5 2142.87    5170 2143.97  5300.2 2148.93  5477.9 2161.07
#Mann= 5 ,-1 , 0
  4726.8     .07       0  4799.7     .16       0  5003.4     .07       0
  5012.2     .16       0  5300.2     .07       0
Bank Sta=5003.4,5012.2
XS Rating Curve= 0 ,0
Exp/Cntr=0.3,0.1

Type RM Length L Ch R = 1 ,20595   ,262,262,262
BEGIN DESCRIPTION:
676
END DESCRIPTION:
XS GIS Cut Line= 3
      1531063.67      6786955.92      1530568.91       6787094.8
      1529983.01      6787316.14
#Sta/Elev= 30
    4482 2180.64  4622.5 2178.44    4678 2175.03  4698.7  2176.3  4719.5 2172.43
  4727.5 2167.82  4732.6 2169.06  4740.3 2163.74  4766.7 2154.09    4813 2146.61
  4823.4  2139.4  4833.8  2136.7  4840.1 2139.65  4854.5  2141.9  4937.6 2133.14
  4952.7  2127.9  4958.4 2122.32  4986.6 2114.87  4987.1 2114.37  4997.4 2114.87
  5047.8 2128.81  5181.8 2128.24    5243 2136.52  5320.8 2139.02  5366.6  2143.1
  5481.1 2156.97    5504 2162.24  5523.5 2160.21  5583.8 2160.04  5622.2 2163.41
#Mann= 5 ,-1 , 0
    4482     .07       0  4622.5     .16       0  4986.6     .07       0
  4997.4     .16       0  5366.6     .07       0
Bank Sta=4986.6,4997.4
XS Rating Curve= 0 ,0
Exp/Cntr=0.3,0.1

Type RM Length L Ch R = 1 ,20333   ,219,219,219
BEGIN DESCRIPTION:
675
END DESCRIPTION:
XS GIS Cut Line= 3
      1530989.89      6786725.89      1530456.07      6786873.45
      1529774.69      6786916.85
#Sta/Elev= 30
    4446 2179.02  4575.6 2180.23  4679.1 2175.01  4701.6 2172.58  4741.6 2154.41
    4752 2151.89  4809.8    2143  4883.6 2135.87  4917.9 2129.43  4923.1 2130.04
  4928.3 2126.82  4949.1 2125.13  4957.4 2122.57  4974.7 2113.44  4975.2 2112.94
  4985.8 2113.44  5010.9 2116.15    5031 2122.56    5051 2126.35  5281.5 2128.24
  5331.6 2138.37  5369.3  2148.8  5381.7 2149.59  5451.8 2161.96  5491.9 2162.06
  5511.9 2159.11    5562 2167.45  5624.6 2172.83  5652.2 2179.33  5682.6 2191.77
#Mann= 5 ,-1 , 0
    4446     .07       0  4679.1     .16       0  4974.7     .07       0
  4985.8     .16       0  5369.3     .07       0
Bank Sta=4974.7,4985.8
XS Rating Curve= 0 ,0
Exp/Cntr=0.3,0.1

Type RM Length L Ch R = 1 ,20114   ,274,274,274
BEGIN DESCRIPTION:
674
END DESCRIPTION:
XS GIS Cut Line= 3
       1530807.6      6786556.62      1530390.96       6786673.8
      1529749.46      6786842.84
#Sta/Elev= 30
  4566.2 2178.21  4758.1 2172.45  4818.2 2167.22  4846.3 2155.28  4890.9 2142.44
  4958.8 2127.01  4992.8 2124.11    5010 2112.58  5010.5 2112.08  5021.1 2112.58
  5038.2 2115.68  5085.5 2116.12  5148.8 2117.21    5196 2124.18    5243 2123.66
  5263.7 2131.71  5269.7 2138.71  5281.6 2145.75  5294.7 2157.54  5304.9 2159.89
    5310  2156.7  5367.1 2164.62  5439.5 2168.15  5466.1  2173.8  5471.3 2170.86
  5506.4  2171.3  5522.2 2177.11  5622.1 2194.87  5646.3 2196.52  5662.4 2201.34
#Mann= 7 ,-1 , 0
  4566.2     .07       0  4758.1     .16       0    5010     .07       0
  5021.1     .16       0  5085.5     .07       0    5196     .16       0
  5281.6     .07       0
Bank Sta=5010,5021.1
XS Rating Curve= 0 ,0
Exp/Cntr=0.3,0.1

Type RM Length L Ch R = 1 ,19840   ,334,334,334
BEGIN DESCRIPTION:
673
END DESCRIPTION:
XS GIS Cut Line= 3
      1530772.91      6786482.82      1530195.65      6786474.14
      1529744.23      6786582.66
#Sta/Elev= 30
  4432.4 2176.92  4550.3 2170.67  4590.3 2154.99  4620.3  2153.5  4657.1 2145.76
    4771 2122.94  4900.4 2123.36  4930.4  2120.7  4950.4 2114.93  4990.4 2113.79
  5015.1 2110.51  5015.6 2110.01  5026.2 2110.51  5041.2 2114.06    5047 2122.41
  5052.1 2122.16  5082.4 2137.29    5089 2144.03  5094.1 2141.42  5113.2 2156.64
  5123.5 2160.05  5226.4 2164.41  5298.4 2162.62  5339.5 2164.57  5380.6 2170.22
  5411.5 2181.54  5429.8 2179.52  5434.9 2182.34  5452.6 2175.38    5474 2173.32
#Mann= 5 ,-1 , 0
  4432.4     .07       0  4657.1     .16       0    4771     .07       0
  5015.1     .07       0  5026.2     .07       0
Bank Sta=5015.1,5026.2
XS Rating Curve= 0 ,0
Exp/Cntr=0.3,0.1

Type RM Length L Ch R = 1 ,19506   ,282,282,282
BEGIN DESCRIPTION:
672
END DESCRIPTION:
XS GIS Cut Line= 3
      1530846.71      6786239.77      1530430.02      6786257.13
      1529988.67      6786036.45
#Sta/Elev= 30
  4588.4 2173.03  4640.2 2171.11  4680.2 2171.67  4750.3 2167.81  4770.3 2164.09
  4809.8  2148.7  4870.4 2123.81  4905.8 2119.84  4920.4 2119.68  4938.9 2114.04
  4950.4 2111.05  4970.4 2109.46  4974.9 2107.05  4975.4 2106.55  4986.1 2107.05
  5044.6 2111.05  5166.6 2112.29  5172.2 2113.34  5194.6  2125.5  5216.9 2125.82
    5256 2129.34  5261.6 2129.29  5273.9 2132.87  5312.9 2142.27  5351.1 2145.77
  5367.9 2151.19  5395.8 2155.95  5402.4 2159.41  5424.7 2161.18  5498.9 2156.88
#Mann= 7 ,-1 , 0
  4588.4     .07       0  4809.8     .16       0  4938.9     .07       0
  4974.9     .07       0  4986.1     .07       0    5256     .16       0
  5273.9     .07       0
Bank Sta=4974.9,4986.1
XS Rating Curve= 0 ,0
Exp/Cntr=0.3,0.1

Type RM Length L Ch R = 1 ,19224   ,231,231,231
BEGIN DESCRIPTION:
671
END DESCRIPTION:
XS GIS Cut Line= 3
      1530916.17      6786165.99      1530456.07      6786018.41
      1530030.74      6785988.03
#Sta/Elev= 30
  4515.4 2170.38  4579.6 2170.98  4657.3 2167.18  4684.2 2154.39  4695.2 2152.92
  4716.2 2158.96  4721.5 2162.96  4726.8 2161.25  4737.2 2165.44  4747.7  2163.2
  4755.7 2158.66  4779.2 2153.29  4785.8 2143.42  4800.2 2132.18  4823.1  2121.2
  4831.7 2119.13  4968.2 2117.42  4978.5 2114.42  4990.9 2104.43  4991.4 2103.93
  5002.1 2104.43  5019.7 2108.51  5059.8 2112.74  5074.7 2120.24  5170.1 2120.91
  5215.1 2124.64  5270.3  2141.9    5293  2146.9  5360.6 2156.01    5425  2160.2
#Mann= 5 ,-1 , 0
  4515.4     .07       0  4755.7     .16       0  4990.9     .07       0
  5002.1     .16       0    5293     .07       0
Bank Sta=4990.9,5002.1
XS Rating Curve= 0 ,0
Exp/Cntr=0.3,0.1

Type RM Length L Ch R = 1 ,18993   ,208,208,208
BEGIN DESCRIPTION:
670
END DESCRIPTION:
XS GIS Cut Line= 3
      1530985.56       6785736.3      1530508.15       6785801.4
      1529950.21      6785983.05
#Sta/Elev= 30
  4514.1 2165.64  4524.9 2167.38  4544.9 2169.84    4555 2168.08  4566.9 2160.58
  4585.3 2156.53  4724.8 2141.95  4756.9 2140.51  4783.9 2133.64    4789 2129.61
  4847.7 2115.33    4878 2113.77  4958.7 2120.92    4989 2117.27    4995 2110.11
  5002.8 2110.18  5004.2 2105.12  5004.7 2104.62  5015.4 2105.12  5125.2 2108.08
  5162.4 2110.99  5167.7 2114.31  5188.5 2115.63  5194.4 2118.96  5251.6 2122.09
  5283.2 2128.31  5322.1 2145.14  5348.8 2147.92    5462 2159.25  5582.7 2155.24
#Mann= 6 ,-1 , 0
  4514.1     .16       0  4524.9     .07       0  4724.8     .16       0
  5004.2     .07       0  5015.4     .16       0  5348.8     .07       0
Bank Sta=5004.2,5015.4
XS Rating Curve= 0 ,0
Exp/Cntr=0.3,0.1

Type RM Length L Ch R = 1 ,18785   ,190,190,190
BEGIN DESCRIPTION:
669
END DESCRIPTION:
XS GIS Cut Line= 3
      1531072.43      6785701.58      1530451.73      6785610.43
      1529709.75      6785523.65
#Sta/Elev= 30
    4374 2166.03  4482.6 2167.96    4523 2158.22  4593.8 2145.78  4644.4 2138.58
  4655.9 2139.08  4684.7 2137.25  4709.2 2128.06  4715.1 2123.42    4779 2113.62
  4856.6 2110.84  4937.4  2111.8  4977.8 2106.81  4983.3 2103.48  4991.6 2102.81
  4992.1 2102.31  5002.8 2102.81    5129  2106.4  5147.7 2110.36  5152.8 2108.12
  5179.3 2116.46  5209.5 2118.19  5264.4 2126.11  5319.4 2141.31  5324.4 2139.24
  5360.5 2143.47  5407.7 2143.23    5572 2155.94  5672.8 2157.12  5748.4 2164.96
#Mann= 5 ,-1 , 0
    4374     .07       0  4655.9     .16       0  4991.6     .07       0
  5002.8     .16       0  5264.4     .07       0
Bank Sta=4991.6,5002.8
XS Rating Curve= 0 ,0
Exp/Cntr=0.3,0.1

Type RM Length L Ch R = 1 ,18595   ,319,319,319
BEGIN DESCRIPTION:
668
END DESCRIPTION:
XS GIS Cut Line= 3
      1531141.83      6785653.83      1530460.41      6785449.84
      1530013.35      6785067.89
#Sta/Elev= 30
  4284.2 2165.65  4301.8 2162.53  4343.5  2162.8  4396.3 2152.38  4424.2 2152.48
  4576.1 2138.08    4594 2136.44  4646.2 2120.64  4709.8 2112.71  4750.6 2109.59
  4802.8  2110.6  4814.3 2107.83  4833.4 2110.18  4880.5 2103.36  4951.9 2105.16
  5001.8 2101.21  5002.3 2100.71  5013.5 2101.21  5039.6 2102.58    5057 2105.27
  5074.8 2112.43  5107.5 2120.32  5149.2 2144.26    5192  2160.5  5227.2 2159.62
  5249.1 2151.99  5277.7 2147.85  5376.5 2152.35    5483 2152.08  5583.5 2161.04
#Mann= 7 ,-1 , 0
  4284.2     .07       0  4576.1     .16       0  4833.4     .07       0
  5001.8     .07       0  5013.5     .07       0  5039.6     .16       0
  5074.8     .07       0
Bank Sta=5001.8,5013.5
XS Rating Curve= 0 ,0
Exp/Cntr=0.3,0.1

Type RM Length L Ch R = 1 ,18276   ,336,336,336
BEGIN DESCRIPTION:
667
END DESCRIPTION:
XS GIS Cut Line= 3
      1531311.11      6785623.45      1530703.46      6785280.57
      1530069.85      6785015.84
#Sta/Elev= 30
  4301.8 2177.68  4405.4 2174.17    4508 2142.37  4632.2 2126.16  4648.1 2129.06
  4653.8  2125.1    4664 2128.85  4669.7 2125.36  4685.7 2129.11  4695.1 2125.87
    4729 2122.09  4750.6 2114.97  4882.9 2108.09  4896.5 2102.88  4905.9 2102.58
  4912.4 2107.34  4971.6  2107.7  5002.8 2099.11  5003.3 2098.61  5014.5 2099.11
  5075.1 2106.87  5146.5  2110.1  5189.9 2121.03  5228.8 2130.04  5276.4 2152.34
  5300.2 2158.88  5483.1 2160.34  5512.3 2164.01  5589.2 2158.57  5686.2 2159.68
#Mann= 5 ,-1 , 0
  4301.8     .07       0  4695.1     .16       0  5002.8     .07       0
  5014.5     .16       0  5189.9     .07       0
Bank Sta=5002.8,5014.5
XS Rating Curve= 0 ,0
Exp/Cntr=0.3,0.1

Type RM Length L Ch R = 1 ,17940   ,187,187,187
BEGIN DESCRIPTION:
666
END DESCRIPTION:
XS GIS Cut Line= 3
      1531376.19      6785402.08      1530924.82      6785085.25
      1530343.23      6784894.29
#Sta/Elev= 30
    4433 2175.11  4465.6 2169.81  4501.3 2171.16  4516.1 2165.76  4522.3 2168.18
  4581.1 2145.12  4623.3 2154.33  4638.2 2149.14    4653 2148.51  4659.1 2152.36
  4673.9  2148.2  4694.8 2154.47  4745.6 2143.42  4861.3 2106.66    4924 2100.22
  4932.7 2104.03    4987 2103.66  4999.5 2096.95    5000 2096.45  5011.2 2096.95
  5091.8 2100.84  5117.9 2110.28  5154.9 2109.53  5213.3 2133.14  5331.6 2134.97
  5404.2 2147.44  5467.8 2150.43  5473.1 2147.23  5536.7 2155.85  5596.6 2158.25
#Mann= 5 ,-1 , 0
    4433     .07       0  4745.6     .16       0  4999.5     .07       0
  5011.2     .16       0  5091.8     .07       0
Bank Sta=4999.5,5011.2
XS Rating Curve= 0 ,0
Exp/Cntr=0.3,0.1

Type RM Length L Ch R = 1 ,17753   ,283,283,283
BEGIN DESCRIPTION:
665
END DESCRIPTION:
XS GIS Cut Line= 3
      1531510.74      6785089.59       1530998.6        6784929.
      1530252.05       6784842.2
#Sta/Elev= 30
  4470.7 2175.25  4581.5 2174.15  4627.5 2167.85    4660 2168.18  4692.4 2172.03
  4717.8 2171.04  4730.1 2169.31  4748.5 2161.63  4770.2 2149.74  4789.7 2141.98
  4794.9 2141.98  4822.1  2127.8  4827.4 2130.01    4833 2123.65  4859.8 2112.89
  4897.5 2105.08  4962.3 2101.21  5000.8 2095.87  5001.3 2095.37  5012.5 2095.87
  5111.7 2098.87  5141.4 2106.23  5146.5 2104.09    5152 2106.87  5174.1 2109.59
  5252.7 2113.52  5333.2 2128.19  5433.9 2136.45  5544.6 2148.95    5759 2161.06
#Mann= 5 ,-1 , 0
  4470.7     .07       0  4748.5     .16       0  5000.8     .07       0
  5012.5     .07       0  5174.1     .07       0
Bank Sta=5000.8,5012.5
XS Rating Curve= 0 ,0
Exp/Cntr=0.3,0.1

Type RM Length L Ch R = 1 ,17470   ,158,158,158
BEGIN DESCRIPTION:
664
END DESCRIPTION:
XS GIS Cut Line= 3
      1531562.82      6784846.54      1530842.35      6784703.31
      1530252.07      6784685.95
#Sta/Elev= 30
  4278.5 2171.85  4327.3 2171.07    4368 2164.72  4396.4 2171.69  4429.2 2168.86
  4510.8 2149.37  4582.1 2145.81  4595.5 2142.43  4600.9 2139.52    4606 2140.56
  4622.9 2127.13    4652 2113.86  4657.1 2115.09  4663.7 2111.76  4694.3 2106.39
  4765.7 2100.61  4786.1 2095.83  4801.2 2097.65  4826.8  2095.3    4837 2099.93
    4895 2100.29    4939 2094.63  4973.9 2093.26  4974.4 2092.76  4985.6 2093.26
  5019.5 2104.77  5130.1 2113.01  5220.5 2133.82  5364.7 2140.94  5603.6 2158.73
#Mann= 7 ,-1 , 0
  4278.5     .07       0  4595.5     .16       0  4801.2     .07       0
    4895     .16       0  4973.9     .07       0  4985.6     .16       0
  5130.1     .07       0
Bank Sta=4973.9,4985.6
XS Rating Curve= 0 ,0
Exp/Cntr=0.3,0.1

Type RM Length L Ch R = 1 ,17312   ,225,225,225
BEGIN DESCRIPTION:
663
END DESCRIPTION:
XS GIS Cut Line= 3
      1531528.11      6784681.61      1530937.84      6784581.78
      1530286.83      6784351.76
#Sta/Elev= 30
  4415.2  2148.2  4491.2 2143.85    4682 2139.46  4734.1 2136.06  4793.6 2130.39
  4803.8 2127.25  4844.3 2125.19  4883.2 2112.26  4888.3  2114.3  4925.5 2098.54
  4943.6 2093.56  4976.2  2095.8  5021.6 2092.05  5022.1 2091.55  5033.4 2092.05
  5048.7 2098.98  5129.2 2107.37  5134.5 2105.72  5165.5 2111.45  5216.7 2114.97
    5222 2113.33  5247.6 2117.63  5252.9 2116.33  5283.8 2123.42  5340.4 2131.08
  5441.1 2136.57  5551.5 2146.55  5589.6 2145.46  5644.2 2150.01  5704.3 2151.86
#Mann= 5 ,-1 , 0
  4415.2     .07       0  4491.2     .16       0  4734.1     .07       0
  5021.6     .07       0  5033.4     .07       0
Bank Sta=5021.6,5033.4
XS Rating Curve= 0 ,0
Exp/Cntr=0.3,0.1

Type RM Length L Ch R = 1 ,17087   ,323,323,323
BEGIN DESCRIPTION:
662
END DESCRIPTION:
XS GIS Cut Line= 3
      1531519.43      6784464.59       1530998.6      6784373.45
      1530529.94      6784308.36
#Sta/Elev= 30
  4478.2 2132.51  4523.3  2133.7  4639.6 2129.57    4706 2129.75  4787.3  2125.1
  4858.3 2128.62  4893.7  2125.6  4919.2 2119.49  4930.1 2114.57  4959.8 2100.36
  4990.3 2097.02  5000.4 2090.78    5007 2089.55  5007.5 2089.05  5018.8 2089.55
  5040.9 2094.22  5061.1 2093.92  5079.5  2098.4  5121.6 2098.37  5206.5  2116.3
  5242.8  2126.2  5283.2 2146.99  5299.6 2152.37  5404.3 2150.18  5434.6 2144.13
    5443 2143.41  5448.1 2145.58  5454.8 2142.91  5464.9 2143.17  5480.1  2150.7
#Mann= 6 ,-1 , 0
  4478.2     .16       0  4639.6     .07       0  4930.1     .16       0
    5007     .07       0  5018.8     .16       0  5206.5     .07       0
Bank Sta=5007,5018.8
XS Rating Curve= 0 ,0
Exp/Cntr=0.3,0.1

Type RM Length L Ch R = 1 ,16764   ,232,232,232
BEGIN DESCRIPTION:
661
END DESCRIPTION:
XS GIS Cut Line= 3
      1531758.15      6784434.21      1531002.94      6784082.65
      1530669.36      6784047.99
#Sta/Elev= 30
  4164.4    2143  4212.2    2139  4381.7 2124.84  4399.1  2118.3  4404.6 2118.42
  4410.5 2113.02  4421.6    2112  4427.5 2119.53    4433 2118.03  4450.4 2123.54
  4455.9 2122.03  4473.3 2125.61  4496.1  2126.8  4547.4 2116.53  4638.9  2113.3
  4855.8 2097.06  4962.1 2095.15    4997 2090.78  4999.5 2088.54    5000 2088.04
  5011.3 2088.54  5090.8 2096.85  5095.9 2101.61  5126.1 2112.14  5154.5 2128.53
  5184.5 2147.74  5189.5 2146.85  5216.5 2156.35  5276.9 2160.05  5332.8 2159.19
#Mann= 5 ,-1 , 0
  4164.4     .07       0  4212.2     .16       0  4999.5     .07       0
  5011.3     .16       0  5154.5     .07       0
Bank Sta=4999.5,5011.3
XS Rating Curve= 0 ,0
Exp/Cntr=0.3,0.1

Type RM Length L Ch R = 1 ,16532   ,257,257,257
BEGIN DESCRIPTION:
660
END DESCRIPTION:
XS GIS Cut Line= 3
      1531766.84       6783904.7      1531163.53      6783935.08
      1530573.24      6783791.85
#Sta/Elev= 30
    4385 2166.13  4426.9 2166.65  4446.7 2159.62  4466.9 2150.53    4497 2143.95
  4546.1  2128.6  4597.1 2121.15  4745.6 2112.98  4797.4 2113.59  4847.4 2111.59
  4877.5 2106.92  4907.5 2099.37  4977.6 2093.85  4989.1 2091.88  4989.3 2088.18
  4989.8 2087.68  5001.3 2088.18  5037.1 2090.41  5059.6 2093.69  5167.6 2095.48
  5311.2 2113.62  5339.9 2117.91  5368.3 2125.99  5388.9 2135.96  5409.5  2141.6
  5423.4 2146.82    5430 2152.04  5450.6 2158.82  5491.8 2161.61  5596.5    2163
#Mann= 5 ,-1 , 0
    4385     .07       0  4446.7     .16       0  4989.3     .07       0
  5001.3     .16       0  5311.2     .07       0
Bank Sta=4989.3,5001.3
XS Rating Curve= 0 ,0
Exp/Cntr=0.3,0.1

Type RM Length L Ch R = 1 ,16275   ,186,186,186
BEGIN DESCRIPTION:
659
END DESCRIPTION:
XS GIS Cut Line= 3
      1531879.67      6783804.87      1531150.51      6783674.66
      1530560.21      6783674.66
#Sta/Elev= 30
  4263.8 2152.89  4327.9 2164.41  4386.8 2166.99  4451.4 2164.85  4461.6 2161.86
  4486.6  2149.5  4512.3 2135.87  4542.8 2123.44  4558.5 2117.58  4583.5 2112.47
  4676.3 2105.26  4715.5 2103.55  4806.9 2094.56    4878 2091.15  4969.5 2091.12
  4979.6 2088.49  4989.8 2083.88  4993.7 2083.88  4994.2 2083.38  5005.7 2083.88
    5010 2089.14    5020 2091.35    5100    2092    5210 2102.68  5267.7 2112.91
    5290 2116.83    5310 2123.03    5390 2159.35    5510 2164.04  5594.8 2165.12
#Mann= 5 ,-1 , 0
  4263.8     .07       0  4486.6     .16       0  4993.7     .07       0
  5005.7     .16       0  5267.7     .07       0
Bank Sta=4993.7,5005.7
XS Rating Curve= 0 ,0
Exp/Cntr=0.3,0.1

Type RM Length L Ch R = 1 ,16089   ,289,289,289
BEGIN DESCRIPTION:
658
END DESCRIPTION:
XS GIS Cut Line= 3
      1531953.51      6783679.01      1531150.51      6783488.03
      1530512.53      6783518.41
#Sta/Elev= 30
  4183.1 2162.67  4250.3 2160.98  4292.5 2155.05  4297.7 2150.95  4334.7 2148.59
  4339.8 2151.76  4376.8 2137.11    4382 2139.86  4407.7 2132.64  4424.2 2132.46
  4429.3 2128.32  4465.3 2123.96  4724.5 2092.16  4945.6  2089.5  4987.6 2084.26
  4988.1 2083.76  4999.6 2084.26  5003.6 2088.92    5014  2090.8  5074.1 2090.99
    5111 2101.57  5167.9 2109.25  5304.3 2128.55  5394.4 2158.66  5464.5 2159.95
  5504.6 2151.69  5531.5 2158.08  5574.6 2154.06  5635.2 2161.08  5647.2 2161.58
#Mann= 6 ,-1 , 0
  4183.1     .07       0  4465.3     .16       0  4987.6     .07       0
  4999.6     .16       0  5167.9     .07       0  5635.2    .035       0
Bank Sta=4987.6,4999.6
XS Rating Curve= 0 ,0
Exp/Cntr=0.3,0.1

Type RM Length L Ch R = 1 ,15800   ,184,184,184
BEGIN DESCRIPTION:
657
END DESCRIPTION:
XS GIS Cut Line= 3
      1531888.38      6783548.81      1531389.23      6783336.12
      1530639.15      6783201.72
#Sta/Elev= 30
  4458.2 2156.04  4505.4 2150.79  4522.9 2155.41  4528.3  2149.9  4546.5 2151.13
  4551.9 2146.35  4570.1 2148.28  4575.5 2142.83  4592.3 2139.57  4631.2 2123.35
  4804.5 2098.95  4918.4 2087.75  4998.1 2087.17  5005.5 2086.92  5008.3 2081.76
  5008.8 2081.26  5020.3 2081.76  5035.6 2088.49  5208.3 2087.59  5269.2  2091.2
  5327.4 2098.51  5367.1 2101.78  5533.6 2118.63    5605 2133.11  5641.1 2142.56
  5646.2 2138.54  5685.7 2149.25  5694.8 2150.49  5699.9 2146.83  5762.8 2156.66
#Mann= 8 ,-1 , 0
  4458.2     .07       0  4631.2     .16       0  4998.1     .07       0
  5008.3     .07       0  5020.3     .07       0  5327.4     .16       0
  5367.1     .07       0    5605    .035       0
Bank Sta=5008.3,5020.3
XS Rating Curve= 0 ,0
Exp/Cntr=0.3,0.1

Type RM Length L Ch R = 1 ,15616   ,295,295,295
BEGIN DESCRIPTION:
14
END DESCRIPTION:
XS GIS Cut Line= 3
      1531855.01      6783388.01      1531496.86      6783194.04
      1530804.99        6782988.
#Sta/Elev= 30
  4592.7 2162.53  4595.6 2162.53  4600.8 2158.55  4650.2 2133.92  4672.3 2125.25
  4726.4 2111.77  4742.9 2111.02  4820.2 2101.33    4830  2101.5  4895.6 2088.93
  4923.2 2085.89  4977.4 2086.71  5005.4 2086.08  5016.8    2084  5017.3  2083.5
  5028.8    2084  5038.6 2087.57  5104.6  2086.6  5158.5 2084.97  5319.6 2088.17
  5600.6    2105    5628  2113.4  5633.8 2118.03    5639 2117.86  5659.3 2126.74
  5666.9 2132.07  5672.1 2132.34  5700.1  2148.4  5705.3 2146.62  5721.9 2153.48
#Mann= 5 ,-1 , 0
  4592.7     .07       0  4742.9     .16       0  5016.8     .07       0
  5028.8     .16       0  5104.6     .07       0
Bank Sta=5016.8,5028.8
XS Rating Curve= 0 ,0
Exp/Cntr=0.3,0.1

Type RM Length L Ch R = 1 ,15321   ,307,307,307
BEGIN DESCRIPTION:
656
END DESCRIPTION:
XS GIS Cut Line= 3
      1532070.63      6783297.05      1531454.33      6782949.84
      1530781.62      6782793.59
#Sta/Elev= 30
  4289.6 2161.73  4330.5 2160.53  4364.9 2154.97  4402.4 2156.18  4418.3 2148.73
  4424.1 2150.73    4440 2143.88  4445.7 2145.86  4477.6  2135.2  4499.3 2129.89
    4505 2130.81  4520.9  2125.4  4639.4 2109.18  4858.5  2091.9  4887.9 2086.39
  4978.7 2082.64  4979.2 2082.14  4990.7 2082.64  4993.8 2085.08  5016.8 2085.93
  5180.1 2084.24  5232.4  2084.6  5305.9  2093.9  5428.8 2093.91  5499.3 2100.36
  5514.1 2103.68  5571.2 2135.39  5604.5 2150.67  5667.6 2152.38  5687.6 2152.07
#Mann= 6 ,-1 , 0
  4289.6     .07       0  4978.7     .07       0  4990.7     .07       0
  5180.1    .035       0  5305.9     .07       0  5667.6    .035       0
Bank Sta=4978.7,4990.7
XS Rating Curve= 0 ,0
Exp/Cntr=0.3,0.1

Type RM Length L Ch R = 1 ,15014   ,276,276,276
BEGIN DESCRIPTION:
655
END DESCRIPTION:
XS GIS Cut Line= 3
      1531931.75      6783080.04      1531358.84      6782672.06
      1530890.13      6782585.26
#Sta/Elev= 30
    4294 2135.61  4342.9 2149.03  4357.7 2141.39  4363.8 2142.27  4387.2 2134.87
  4393.3 2136.41  4408.1 2129.61    4429 2129.52  4458.5 2121.19  4486.4 2121.25
  4494.2 2116.92    4536  2105.7  4572.8 2098.85    4788 2083.66  4940.1 2083.66
    4981 2083.38  4983.6 2080.02  4984.1 2079.52  4995.7 2080.02  4995.8 2082.91
  5001.8 2083.69  5021.6 2082.57  5104.6 2087.67  5230.4 2093.85  5316.5 2101.85
  5367.4 2122.43    5408 2142.33  5418.2 2144.36  5432.5 2145.21    5474  2139.2
#Mann= 7 ,-1 , 0
    4294     .07       0  4572.8     .16       0  4940.1     .07       0
  4983.6     .07       0  4995.7     .07       0  5104.6    .035       0
  5230.4     .07       0
Bank Sta=4983.6,4995.7
XS Rating Curve= 0 ,0
Exp/Cntr=0.3,0.1

Type RM Length L Ch R = 1 ,14738   ,166,166,166
BEGIN DESCRIPTION:
654
END DESCRIPTION:
XS GIS Cut Line= 3
      1532153.09       6782871.7      1531406.59      6782411.64
      1530895.71      6782212.49
#Sta/Elev= 30
  4121.1  2146.1  4137.1  2153.4  4179.6 2153.72    4195  2149.9  4231.7 2134.81
  4289.7 2121.43  4326.3 2119.85  4332.2 2122.36  4384.3 2123.62  4405.6 2127.04
    4421 2124.18  4426.9 2126.05  4471.2 2118.13  4484.8 2109.83  4515.6 2101.55
  4631.5 2090.45  4745.1 2082.97  4793.4 2079.95  4793.9 2079.45  4805.7 2079.95
  5092.2 2081.61  5127.5 2091.65  5171.4 2096.72  5203.6 2104.76  5235.8 2115.76
    5252 2124.75  5266.1 2129.96  5278.7  2138.1  5301.3 2140.55  5546.3 2146.45
#Mann= 7 ,-1 , 0
  4121.1     .07       0  4631.5     .16       0  4745.1     .07       0
  4793.4     .07       0  4805.7     .07       0  5092.2     .16       0
    5252     .07       0
Bank Sta=4793.4,4805.7
XS Rating Curve= 0 ,0
Exp/Cntr=0.3,0.1

Type RM Length L Ch R = 1 ,14572   ,339,339,339
BEGIN DESCRIPTION:
653
END DESCRIPTION:
XS GIS Cut Line= 3
      1532344.04      6782541.84      1531410.93      6782246.71
      1530934.94      6782112.57
#Sta/Elev= 30
  4014.5 2132.14    4047 2130.15  4065.9 2131.07  4138.7 2124.39  4149.8 2121.89
  4170.8 2122.46  4208.6 2119.27  4213.8 2120.58    4261 2116.96  4273.2 2112.67
  4278.4 2115.02  4305.5 2108.35  4412.9 2095.57  4707.7 2080.84  4779.1 2078.98
  4861.1 2080.45  4940.9  2081.1  4999.3 2081.17  4999.5 2078.55    5000 2078.05
  5011.8 2078.55  5030.5 2080.03  5044.9 2085.12  5051.3 2092.01  5072.1 2096.53
  5134.4 2116.57  5157.3 2119.53  5196.7 2138.02    5377 2139.59  5487.7    2144
#Mann= 7 ,-1 , 0
  4014.5     .07       0    4261     .16       0  4707.7     .07       0
  4861.1     .16       0  4940.9     .07       0  4999.5     .07       0
  5011.8     .07       0
Bank Sta=4999.5,5011.8
XS Rating Curve= 0 ,0
Exp/Cntr=0.3,0.1

Type RM Length L Ch R = 1 ,14233   ,157,157,157
BEGIN DESCRIPTION:
652
END DESCRIPTION:
XS GIS Cut Line= 3
      1532482.93      6782368.22       1531580.2      6782047.06
      1531150.52      6781843.07
#Sta/Elev= 30
  4052.5 2141.85  4092.7 2133.99  4103.4 2129.58  4167.1  2119.8    4380 2103.91
  4496.1 2096.82  4606.3 2093.48  4643.7 2097.96  4693.5 2094.68  4761.4 2084.58
  4842.4 2079.02  4898.8 2077.43  4956.6 2079.18  4984.3 2080.56  4996.6 2078.01
    5021  2080.8  5128.5 2077.41    5129 2076.91  5140.9 2077.41  5157.4 2080.08
  5176.9 2088.92  5215.7 2106.47  5231.1 2111.37  5259.9  2126.3  5276.6 2131.87
  5305.5 2131.32  5344.8  2125.6  5357.8 2129.41  5381.7 2132.96  5486.3 2137.42
#Mann= 9 ,-1 , 0
  4052.5     .07       0    4380     .16       0  4643.7     .07       0
  4956.6     .16       0  5128.5     .07       0  5140.9     .16       0
  5176.9     .07       0  5305.5     .16       0  5357.8     .07       0
Bank Sta=5128.5,5140.9
XS Rating Curve= 0 ,0
Exp/Cntr=0.3,0.1

Type RM Length L Ch R = 1 ,14076   ,199,199,199
BEGIN DESCRIPTION:
651
END DESCRIPTION:
XS GIS Cut Line= 3
      1532443.89      6782168.58      1531610.58      6781899.49
      1531141.79      6781795.32
#Sta/Elev= 30
  4117.9 2144.83  4139.5 2143.22  4166.3 2137.38  4171.6 2138.71  4203.6 2127.73
  4211.3 2123.14  4230.4 2121.66  4235.6 2118.18  4274.4 2109.49  4331.7 2106.22
  4363.8 2101.74  4377.4 2102.33  4513.8 2094.06  4568.6 2095.77  4642.2 2083.44
  4778.8 2081.18  4835.6 2076.05  4836.1 2075.55    4848 2076.05  4935.7 2079.19
  5091.5 2077.91  5142.7 2083.93  5159.9 2091.75  5165.1 2090.54  5175.2 2095.43
  5203.5 2107.41  5208.6  2107.3  5214.4 2111.99  5252.1 2129.48  5473.8  2141.3
#Mann= 7 ,-1 , 0
  4117.9     .07       0  4377.4     .16       0  4513.8     .07       0
  4835.6     .07       0    4848     .07       0  4935.7     .16       0
  5175.2     .07       0
Bank Sta=4835.6,4848
XS Rating Curve= 0 ,0
Exp/Cntr=0.3,0.1

Type RM Length L Ch R = 1 ,13877   ,312,312,312
BEGIN DESCRIPTION:
650
END DESCRIPTION:
XS GIS Cut Line= 3
      1532456.91      6782047.05      1531549.82      6781712.86
      1531129.37      6781613.16
#Sta/Elev= 30
  4039.1 2122.59  4109.5 2116.46  4195.6 2117.16  4211.6 2111.13  4256.4 2106.83
  4281.6 2100.78    4312 2104.55  4337.1 2092.81  4342.5 2096.59  4350.2 2096.93
  4367.6  2091.2  4392.7 2088.35  4484.1    2088  4520.7 2082.68  4611.4 2078.42
  4710.8 2075.18  4711.3 2074.68  4723.2 2075.18    4803 2078.74  5000.2 2077.38
  5082.7 2084.23  5120.5 2097.27  5185.5 2128.24  5207.3 2127.29  5236.8 2131.72
  5289.4 2133.54  5329.3 2132.88  5390.6 2138.53  5395.7 2136.16  5437.9 2142.76
#Mann= 7 ,-1 , 0
  4039.1     .07       0  4611.4     .16       0  4710.8     .07       0
  4723.2     .16       0  5120.5     .07       0  5207.3    .035       0
  5289.4     .07       0
Bank Sta=4710.8,4723.2
XS Rating Curve= 0 ,0
Exp/Cntr=0.3,0.1

Type RM Length L Ch R = 1 ,13565   ,267,267,267
BEGIN DESCRIPTION:
649
END DESCRIPTION:
XS GIS Cut Line= 3
      1532361.41      6781851.73      1531714.75      6781456.78
      1531315.42      6781339.59
#Sta/Elev= 30
  4234.5 2130.61  4277.2 2136.36  4292.2 2130.86  4307.6 2119.76  4328.9 2114.41
  4359.2 2100.88  4381.2 2100.37  4429.6 2106.14  4460.5 2094.85  4481.8 2095.06
  4545.6 2082.16  4729.6 2074.25  4738.8 2071.23  4739.3 2070.73  4751.2 2071.23
    4781 2074.94  4994.7 2074.22  5012.8  2077.7  5066.8 2078.63  5127.5 2080.82
  5200.4 2090.18  5222.6 2093.78  5250.8  2103.5    5256 2102.23  5289.4  2117.6
  5294.6 2116.65  5322.8  2126.9  5367.2 2131.65  5404.5 2131.59  5408.4 2131.45
#Mann= 6 ,-1 , 0
  4234.5     .07       0  4545.6     .16       0  4738.8     .07       0
  4751.2     .16       0  5066.8     .07       0  5404.5    .035       0
Bank Sta=4738.8,4751.2
XS Rating Curve= 0 ,0
Exp/Cntr=0.3,0.1

Type RM Length L Ch R = 1 ,13298   ,192,192,192
BEGIN DESCRIPTION:
648
END DESCRIPTION:
XS GIS Cut Line= 3
      1532378.84       6781799.7      1531784.19      6781213.73
      1531636.61      6781027.08
#Sta/Elev= 30
  4162.7 2121.06  4173.7 2122.52  4180.8 2127.05  4194.9 2130.65  4209.1 2129.06
  4251.5 2117.19  4350.5 2105.89  4371.7 2101.29  4378.7 2096.86  4392.8 2093.13
  4484.8 2078.42    4515 2076.47  4563.9 2073.21  4612.1 2072.49  4620.1 2070.52
  4620.6 2070.02  4632.5 2070.52  4640.4 2072.72  4684.9 2072.63  4746.4 2072.24
  4760.6 2074.79  5015.8 2072.36  5065.5 2074.81  5144.1 2085.84  5164.9 2092.37
  5171.2  2096.6  5179.3 2097.18  5193.7 2102.57    5234 2120.27  5235.5 2120.27
#Mann= 7 ,-1 , 0
  4162.7     .07       0    4515     .16       0  4563.9     .07       0
  4620.1     .07       0  4632.5     .07       0  4684.9     .16       0
    5234     .07       0
Bank Sta=4620.1,4632.5
XS Rating Curve= 0 ,0
Exp/Cntr=0.3,0.1

Type RM Length L Ch R = 1 ,13106   ,156,156,156
BEGIN DESCRIPTION:
647
END DESCRIPTION:
XS GIS Cut Line= 3
      1532708.66      6781673.79      1531944.78      6781118.24
      1531771.17      6780914.25
#Sta/Elev= 30
  4040.9 2088.49  4262.5 2089.49  4312.8 2097.72  4413.2  2102.5  4441.1 2099.43
  4484.3 2080.26  4497.4  2077.1  4517.8 2073.42  4570.1 2070.01    4706 2070.98
  4812.8 2071.55  4821.3 2069.15  4821.8 2068.65  4833.7 2069.15  4849.1 2071.17
  4877.7 2069.64  4898.6 2072.74  4992.6 2070.66  5077.7 2072.53  5119.9 2077.88
  5148.5 2085.38  5156.2 2091.47  5191.5 2109.16  5197.9 2109.21  5205.6 2115.18
  5212.2 2115.05  5219.9 2121.36  5226.5 2121.43  5234.2 2126.61  5253.3 2129.53
#Mann= 7 ,-1 , 0
  4040.9     .07       0  4497.4     .16       0  4517.8     .07       0
    4706     .16       0  4821.3     .07       0  4833.7     .16       0
  5191.5     .07       0
Bank Sta=4821.3,4833.7
XS Rating Curve= 0 ,0
Exp/Cntr=0.3,0.1

Type RM Length L Ch R = 1 ,12950   ,200,200,200
BEGIN DESCRIPTION:
646
END DESCRIPTION:
XS GIS Cut Line= 3
      1533125.34      6781192.02      1532009.89      6780975.01
      1531876.93       6780902.1
#Sta/Elev= 30
  3856.6  2093.6    3969 2093.32  4006.6 2090.86  4011.7 2092.43  4058.3 2087.28
  4063.4  2090.9  4071.4 2089.53  4109.9  2078.2    4115 2079.17    4132 2074.85
  4378.4 2073.17  4486.9    2070  4556.8 2069.06  4594.4    2067  4594.9  2066.5
  4606.8    2067  4875.7 2068.31  4894.9 2070.83  4906.3 2068.77  4936.8 2070.89
  5000.7 2070.05  5009.9 2071.36  5044.3 2088.41  5076.5 2100.72  5082.2 2105.16
  5098.3  2110.2  5103.1 2114.11  5120.1 2120.72  5125.8 2125.22  5144.6 2128.17
#Mann= 7 ,-1 , 0
  3856.6     .07       0  4071.4     .16       0  4486.9     .07       0
  4556.8     .16       0  4594.4     .07       0  4606.8     .16       0
  5103.1     .07       0
Bank Sta=4594.4,4606.8
XS Rating Curve= 0 ,0
Exp/Cntr=0.3,0.1

Type RM Length L Ch R = 1 ,12750   ,127,127,127
BEGIN DESCRIPTION:
13
END DESCRIPTION:
XS GIS Cut Line= 3
      1533188.71      6781007.13      1532105.43      6780808.18
      1531905.04      6780837.99
#Sta/Elev= 30
  3898.6 2100.52    3943    2108  3977.7 2103.56  3993.9 2098.67  4024.4 2099.47
    4065 2092.59  4083.9 2092.72    4089 2087.48  4115.9 2086.56  4142.1 2081.08
  4147.2  2083.9  4166.7 2078.55  4248.4 2073.46  4534.1 2068.54  4776.8 2067.32
  4790.9 2065.49  4791.4 2064.99  4803.3 2065.49  4842.3 2067.97  4873.1 2068.14
  4949.6 2070.61  5064.9 2070.42  5081.3  2072.9  5103.7 2080.63  5131.9 2097.34
  5162.2 2111.65    5168 2116.73    5173 2116.02  5192.5 2125.41  5202.6 2126.63
#Mann= 7 ,-1 , 0
  3898.6     .07       0  4248.4     .16       0  4790.9     .07       0
  4803.3     .16       0  4842.3     .07       0  4873.1     .16       0
  5064.9     .07       0
Bank Sta=4790.9,4803.3
XS Rating Curve= 0 ,0
Exp/Cntr=0.3,0.1

Type RM Length L Ch R = 1 ,12623   ,231,231,231
BEGIN DESCRIPTION:
645
END DESCRIPTION:
XS GIS Cut Line= 3
       1533112.3      6780714.59      1532109.71      6780679.87
      1531875.38      6780749.31
#Sta/Elev= 30
  3992.4 2083.04  4036.6 2080.74  4041.6 2083.69  4059.7 2080.79  4089.8 2080.71
  4099.8 2082.31  4119.8 2091.19  4149.8 2078.16  4188.7 2076.26    4410    2068
  4710.1 2065.67  4871.2 2067.77  4920.3 2066.53  4930.3 2068.64  4944.1 2064.78
  4944.6 2064.28  4956.5 2064.78  4970.3 2068.87  4990.5 2068.77  5001.8 2067.96
  5044.6 2069.76  5072.7 2082.91  5077.9 2080.72  5111.1 2100.24  5116.3  2098.4
  5144.4 2114.66  5149.6 2112.59    5157 2116.23  5177.6 2119.93    5240 2118.53
#Mann= 7 ,-1 , 0
  3992.4     .07       0  4188.7     .16       0  4871.2     .07       0
  4944.1     .07       0  4956.5     .07       0  4990.5     .16       0
  5001.8     .07       0
Bank Sta=4944.1,4956.5
XS Rating Curve= 0 ,0
Exp/Cntr=0.3,0.1

Type RM Length L Ch R = 1 ,12392   ,161,161,161
BEGIN DESCRIPTION:
644
END DESCRIPTION:
XS GIS Cut Line= 3
       1533125.3      6780323.97      1532166.14      6780458.52
      1531853.63      6780658.17
#Sta/Elev= 30
  4018.2 2114.81  4180.1 2120.09  4226.3 2105.73  4231.4 2107.55  4331.5 2082.75
  4392.1 2085.53  4493.1 2065.78  4646.3 2063.53  4937.4 2065.44  4977.8  2064.6
  4994.3 2060.15  4994.8 2059.65  5006.7 2060.15  5030.9 2063.23  5052.1 2061.37
  5059.3 2065.96  5109.6  2069.4  5124.8 2074.69  5130.8 2079.94  5197.6  2099.9
  5203.5 2104.15  5212.8 2104.12  5218.7 2109.69    5234 2109.19  5239.9  2112.6
  5255.1 2107.67    5261 2110.38  5270.3  2107.7  5312.6 2118.17  5357.6 2116.62
#Mann= 4 ,-1 , 0
  4018.2     .07       0  4646.3     .16       0  4994.3     .07       0
  5006.7     .07       0
Bank Sta=4994.3,5006.7
XS Rating Curve= 0 ,0
Exp/Cntr=0.3,0.1

Type RM Length L Ch R = 1 ,12231   ,377,377,377
BEGIN DESCRIPTION:
643
END DESCRIPTION:
XS GIS Cut Line= 3
      1532795.49      6779942.01      1532053.29      6780363.03
      1531671.86      6780653.44
#Sta/Elev= 30
  4149.2 2115.68  4190.9 2119.05  4223.1 2114.46  4277.4 2089.05  4336.5 2065.56
  4398.6  2060.7  4407.9 2060.27  4476.9 2057.87  4477.4 2057.37  4489.4 2057.87
  4783.7 2063.24  5004.6 2063.37  5022.4 2060.71  5033.6 2058.16    5069 2058.77
  5075.8 2065.46  5089.8 2072.07  5183.3  2080.6  5218.7  2088.1    5254 2090.58
  5276.8 2085.23  5283.1 2088.71  5297.7    2084  5303.9 2086.96  5326.7 2085.17
    5333 2088.45  5347.6 2085.51  5382.9 2091.73  5453.6 2116.22  5481.9 2116.82
#Mann= 7 ,-1 , 0
  4149.2     .07       0  4223.1     .16       0  4398.6     .07       0
  4407.9     .16       0  4476.9     .07       0  4489.4     .16       0
  5022.4     .07       0
Bank Sta=4476.9,4489.4
XS Rating Curve= 0 ,0
Exp/Cntr=0.3,0.1
