--- Indian Creek.prj (project) ---

Proj Title=Indian Creek Base Level Engineering
Current Plan=p01
Default Exp/Contr=0.3,0.1
English Units
Geom File=g01
Flow File=f01
Plan File=p01
Y Axis Title=Elevation
X Axis Title(PF)=Main Channel Distance
X Axis Title(XS)=Station
BEGIN DESCRIPTION:
Indian Creek
END DESCRIPTION:
DSS Export Rating Curves= 0
DSS Export Rating Curve Sorted= 0
DSS Export Volume Flow Curves= 0
DXF OffsetX= 0
DXF OffsetY= 0
DXF ScaleX= 1
DXF ScaleY= 10

--- Indian Creek.p01 (plan) ---

Plan Title=Multiple Run
Program Version=4.10
Short Identifier=Multiple
Geom File=g01
Flow File=f01
Subcritical Flow
K Sum by GR= 0
Std Step Tol= 0.01
Critical Tol= 0.01
Num of Std Step Trials= 20
Max Error Tol= 0.3
Flow Tol Ratio= 0.001
Split Flow NTrial= 30
Split Flow Tol= 0.02
Split Flow Ratio= 0.02
Log Output Level= 0
Friction Slope Method= 1
Unsteady Friction Slope Method= 2
Unsteady Bridges Friction Slope Method= 1
Parabolic Critical Depth
Global Vel Dist= 1 , 1 , 1
Global Log Level= 0
CheckData=True
Encroach Param=-1 ,0,0, 0
BEGIN DESCRIPTION:
Multiple Run
END DESCRIPTION:
Computation Interval=1HOUR
Output Interval=1HOUR
Run HTab= 0
Run UNet= 0
Run PostProcess= 0
Run WQNet= 0
UNET Theta= 1
UNET Theta Warmup= 1
UNET ZTol= 0.02
UNET ZSATol= 0.05
UNET MxIter= 20
UNET MaxInSteps= 0
UNET DtIC= 0
UNET DtMin= 0
UNET MaxCRTS= 20
UNET WFStab= 2
UNET SFStab= 1
UNET WFX= 1
UNET SFX= 1
UNET DSS MLevel= 4
UNET DZMax Abort= 100
UNET Convert EG Bridges= 0
UNET Use Existing IB Tables=-1
UNET Froude Reduction=False
UNET Froude Limit= 1
UNET Froude Power= 10
UNET Time Slicing=0,0, 5
UNET Junction Losses=0
Instantaneous Interval=1HOUR
Write IC File= 0
Write IC File at Sim End=0
Echo Input=False
Echo Parameters=False
Echo Output=False
Write Detailed= 0
WQ AD Non Conservative
WQ ULTIMATE=-1
WQ Max Comp Step=1HOUR
WQ Output Interval=15MIN
WQ Output Selected Increments= 0
WQ Output face flow=0
WQ Output face velocity=0
WQ Output face area=0
WQ Output face dispersion=0
WQ Output cell volume=0
WQ Output cell surface area=0
WQ Output cell continuity=0
WQ Output cumulative cell continuity=0
WQ Output face conc=0
WQ Output face dconc_dx=0
WQ Output face courant=0
WQ Output face peclet=0
WQ Output face adv mass=0
WQ Output face disp mass=0
WQ Output cell mass=0
WQ Output cell source sink temp=0
WQ Output cell source sink nsm=0
WQ Output MaxMinRange=-1
WQ Daily Max Min Mean=-1
WQ Daily Range=0
WQ Daily Time=0
WQ Create Restart=0
WQ Fixed Restart=0
WQ System Summary=0
WQ Use Fixed Temperature=0
Sorting and Armoring Iterations= 10
XS Update Threshold= 0.02
Hydraulics Update Threshold= 0.02
Energy Slope Method= 1
Volume Change Method= 0
XS Weighting Method= 0
Number of US Weighted Cross Sections= 1
Number of DS Weighted Cross Sections= 1
Upstream XS Weight=0.25
Main XS Weight=0.5
Downstream XS Weight=0.25
Number of DS XS's Weighted with US Boundary= 1
Upstream Boundary Weight= 1
Weight of XSs Associated with US Boundary= 0
Number of US XS's Weighted with DS Boundary= 1
Downstream Boundary Weight= 0.5
Weight of XSs Associated with DS Boundary= 0.5
Sediment Output Level= 4
Mass or Volume Output= 0
Output Increment Type= 1
Profile and TS Output Increment= 10
XS Output Flag= 0
XS Output Increment= 10
Disregard all LS=0
Disregard all Conn=0
Disregard all Breaches=0
Disregard all Pumps=0

--- Indian Creek.f01 (steady flow) ---

Flow Title=Multiple
Number of Profiles=7
Profile Names=10-year,25-year,50-year,1pct_min,100-year,1pct_plu,500-year
River Rch & RM= Indian Creek,Reach-1,51296
     260     357     436     330     529     727     787
River Rch & RM= Indian Creek,Reach-1,46204
     359     501     619     474     759    1040    1160
River Rch & RM= Indian Creek,Reach-1,41044
     458     648     808     622     997    1370    1540
River Rch & RM= Indian Creek,Reach-1,37285
     549     784     983     761    1220    1680    1910
River Rch & RM= Indian Creek,Reach-1,33551
     631     906    1140     887    1420    1960    2240
River Rch & RM= Indian Creek,Reach-1,29279
     691     996    1260     980    1570    2160    2480
River Rch & RM= Indian Creek,Reach-1,24516
     752    1090    1370    1070    1720    2370    2730
River Rch & RM= Indian Creek,Reach-1,19184
     831    1210    1530    1200    1920    2640    3060
River Rch & RM= Indian Creek,Reach-1,16431
     892    1300    1650    1290    2070    2840    3300
River Rch & RM= Indian Creek,Reach-1,10018
    1150    1690    2170    1710    2730    3760    4420
River Rch & RM= Indian Creek,Reach-1,7070
    1220    1790    2290    1800    2890    3970    4650
River Rch & RM= Indian Creek,Reach-1,1660
    1260    1840    2360    1860    2980    4090    4810
Boundary for River Rch & Prof#=Indian Creek,Reach-1,1
Up Type=0
Dn Type=3
Dn Slope=0.0002
Boundary for River Rch & Prof#=Indian Creek,Reach-1,2
Up Type=0
Dn Type=3
Dn Slope=0.0002
Boundary for River Rch & Prof#=Indian Creek,Reach-1,3
Up Type=0
Dn Type=3
Dn Slope=0.0002
Boundary for River Rch & Prof#=Indian Creek,Reach-1,4
Up Type=0
Dn Type=3
Dn Slope=0.0002
Boundary for River Rch & Prof#=Indian Creek,Reach-1,5
Up Type=0
Dn Type=3
Dn Slope=0.0002
Boundary for River Rch & Prof#=Indian Creek,Reach-1,6
Up Type=0
Dn Type=3
Dn Slope=0.0002
Boundary for River Rch & Prof#=Indian Creek,Reach-1,7
Up Type=0
Dn Type=3
Dn Slope=0.0002

--- Indian Creek.g01 (geometry) ---

Geom Title=Existing Conditions
Program Version=4.10

River Reach=Indian Creek    ,Reach-1
Reach XY= 30
        1537405.        6841688.      1537847.31      6842384.33
      1537707.07      6843532.53      1538651.46      6844689.47
      1538860.34      6846090.74      1540588.58       6847471.2
      1541137.87      6848571.97      1542496.82      6849381.96
      1543252.83      6851043.43      1543406.85      6852976.86
      1543913.16      6853584.62      1546114.65      6854536.64
      1547958.67      6854430.31      1548425.05      6854087.39
      1548932.24      6854638.29        1550005.      6854145.08
      1550908.42      6854430.21      1552706.47      6853141.54
       1553994.5      6853089.22      1555838.71      6854321.29
      1557256.68       6856784.9      1559344.83       6857138.5
      1560520.21      6856738.51      1562203.53      6856891.56
      1564098.92      6858179.91       1565647.1      6858390.91
      1565760.47      6859082.74      1567110.97      6860135.67
      1569984.97      6859938.04        1572305.        6861088.

Type RM Length L Ch R = 1 ,51296   ,231,231,231
BEGIN DESCRIPTION:
Indian Creek 51295.72
END DESCRIPTION:
XS GIS Cut Line= 3
       1537011.5      6842419.73      1537839.59       6842398.9
      1538579.15      6842471.81
#Sta/Elev= 30
  4168.8 1848.99  4232.3 1847.94  4602.4 1848.26  4762.5 1847.16  4782.5 1847.61
  4822.5 1846.28  4870.4 1846.15  4882.5 1845.59  4942.5 1845.47  4962.5 1844.32
  4997.1 1845.51  5002.6 1846.26  5012.6 1843.92  5020.7 1843.35  5020.9 1842.85
  5024.4 1842.85  5024.7 1843.35  5032.7 1843.54  5043.4 1845.78  5062.9 1846.55
    5083 1845.86  5223.7 1847.42  5263.8 1846.59    5347 1847.07  5394.5 1848.13
  5443.2 1848.04  5454.8 1848.64  5498.4 1848.06  5597.6 1848.36  5740.3 1848.69
#Mann= 6 ,-1 , 0
  4168.8    .035       0  4870.4    .045       0  5020.7    .045       0
  5024.7    .045       0  5498.4     .07       0  5597.6    .045       0
Bank Sta=5020.7,5024.7
XS Rating Curve= 0 ,0
Exp/Cntr=0.3,0.1

Type RM Length L Ch R = 1 ,51065   ,139,139,139
BEGIN DESCRIPTION:
Indian Creek 18.0
END DESCRIPTION:
XS GIS Cut Line= 4
      1537031.69      6842474.87      1537755.67      6842586.45
      1537812.15      6842637.64      1538661.97      6842643.63
#Sta/Elev= 30
  4231.1 1848.37  4248.8 1848.41  4315.4 1847.37  4413.6 1847.77  4649.3 1846.95
  4681.5 1845.99    4749 1846.35  4790.9  1845.5  4821.3 1846.57    4882 1845.35
  4932.6  1843.2  4942.4 1841.99  4942.6 1841.49  4946.4 1841.99  4952.8 1844.59
  4960.8  1846.6  4966.5  1846.6  4971.4 1848.77  4978.2 1847.71  4985.6 1848.73
  4992.4 1848.24  5028.2  1849.6    5035 1847.39  5043.8 1847.59  5072.7  1845.1
  5092.7 1844.41  5263.8 1844.71  5402.7 1846.29  5797.4 1848.16  5889.7  1847.9
#Mann= 7 ,-1 , 0
  4231.1     .07       0  4248.8    .045       0    4749     .07       0
  4942.4     .07       0  4946.4     .07       0  5263.8    .045       0
  5797.4    .035       0
Bank Sta=4942.4,4946.4
XS Rating Curve= 0 ,0
Exp/Cntr=0.3,0.1

Type RM Length L Ch R = 1 ,50926   ,274,274,274
BEGIN DESCRIPTION:
Indian Creek 50913.12
END DESCRIPTION:
XS GIS Cut Line= 3
      1537092.24      6842612.58      1537669.24      6842712.26
      1538605.52      6842890.29
#Sta/Elev= 30
  4376.4 1847.69  4480.7 1846.74  4582.2 1847.35  4632.9 1846.26  4744.5 1846.59
  4830.5 1845.01  4876.5 1846.31  4886.6 1845.15  4947.5  1844.5    4978 1842.99
  4986.2 1840.59  4986.4 1840.09  4990.2 1840.59  4998.3 1842.37    5013 1842.78
  5120.5 1844.27  5183.4 1844.56  5191.8  1843.8    5263 1845.03  5331.3 1844.76
  5449.5 1846.06    5548 1845.71    5559 1846.89  5578.6 1846.64  5606.2 1847.98
  5629.5 1847.23  5658.4  1847.9  5670.2 1846.92  5761.8 1847.67    5915 1846.82
#Mann= 7 ,-1 , 0
  4376.4    .045       0  4830.5     .07       0  4947.5     .16       0
  4986.2     .07       0  4990.2     .16       0    5013     .07       0
  5331.3    .045       0
Bank Sta=4986.2,4990.2
XS Rating Curve= 0 ,0
Exp/Cntr=0.3,0.1

Type RM Length L Ch R = 1 ,50652   ,343,343,343
BEGIN DESCRIPTION:
Indian Creek 50652.24
END DESCRIPTION:
XS GIS Cut Line= 3
      1537105.21      6842987.44      1537704.17       6842961.4
       1538561.8      6842945.81
#Sta/Elev= 30
    4399 1845.73  4769.1 1844.81  4809.2 1845.76  4819.2 1844.58    4826 1844.55
  4839.2 1844.13  4849.2 1844.62  4889.3 1843.15  4899.3 1843.77  4919.3 1842.77
  4969.3 1842.81  4996.4 1841.43  5019.4 1841.56  5024.4 1840.68  5027.3 1840.17
  5027.6 1839.67  5031.2 1839.67  5031.4 1840.17  5039.4 1842.01  5059.4 1842.61
  5099.4 1842.19  5123.5 1842.67  5169.4 1842.66  5199.4 1843.37  5222.5 1842.56
  5409.4  1844.3  5489.4 1844.14  5579.5 1845.73  5719.5 1845.34  5856.3 1846.55
#Mann= 7 ,-1 , 0
    4399    .045       0    4826     .16       0  5024.4     .07       0
  5027.3     .07       0  5031.4     .07       0  5123.5     .16       0
  5222.5    .045       0
Bank Sta=5027.3,5031.4
XS Rating Curve= 0 ,0
Exp/Cntr=0.3,0.1

Type RM Length L Ch R = 1 ,50309   ,253,253,253
BEGIN DESCRIPTION:
Indian Creek 50287.88
END DESCRIPTION:
XS GIS Cut Line= 3
      1537126.02      6843294.73      1537844.29      6843288.24
      1538579.14      6843237.44
#Sta/Elev= 30
  4371.3 1844.04  4570.3 1844.07  4620.3 1843.77  4680.3 1844.33  4845.2 1842.88
  4870.3 1842.76  4890.3 1843.24  4900.3 1843.87  4910.3  1843.7  4920.3 1842.37
  4930.3 1842.05  4940.3 1842.84  4950.3 1842.49  4960.3 1842.99  4980.3  1841.6
  5010.3 1840.41  5040.3 1840.59  5050.3  1841.1  5078.3 1840.24  5078.5 1839.74
  5082.1 1839.74  5082.4 1840.24  5203.6 1840.98  5240.7 1841.44  5290.8 1842.64
  5411.1 1842.67  5511.3 1844.05  5621.6 1843.76  5761.9 1845.67  5826.2 1845.31
#Mann= 5 ,-1 , 0
  4371.3    .045       0  4845.2     .07       0  5078.3     .07       0
  5082.4     .07       0  5203.6    .045       0
Bank Sta=5078.3,5082.4
XS Rating Curve= 0 ,0
Exp/Cntr=0.3,0.1

Type RM Length L Ch R = 1 ,50056   ,439,439,439
BEGIN DESCRIPTION:
Indian Creek 49837.92
END DESCRIPTION:
XS GIS Cut Line= 4
      1537056.95      6843489.17      1537791.72      6843531.34
      1537853.61      6843547.83      1538585.63      6843603.91
#Sta/Elev= 30
  4349.2 1843.36  4497.5  1843.9  4737.9 1842.65    4788 1841.52  4888.1  1841.7
  4936.4 1840.15  4986.3  1839.6  4986.5  1839.1  4990.4  1839.6  4993.2 1839.65
  5028.4 1839.71  5048.4 1840.47  5068.4 1839.81  5078.5 1840.82  5084.3 1843.54
  5088.4 1843.54  5092.7 1841.42  5098.9 1843.58  5109.3 1845.11  5127.6 1845.18
  5132.8 1843.85  5170.7 1843.41  5180.7 1842.08  5216.4 1840.03  5221.4 1841.99
  5250.9 1842.04    5281 1839.93  5301.1 1840.81  5364.7 1840.87  5883.4 1843.84
#Mann= 5 ,-1 , 0
  4349.2    .045       0  4986.3     .07       0  4990.4    .045       0
  4993.2     .07       0  5364.7    .045       0
Bank Sta=4986.3,4990.4
XS Rating Curve= 0 ,0
Exp/Cntr=0.3,0.1

Type RM Length L Ch R = 1 ,49617   ,565,565,565
BEGIN DESCRIPTION:
Indian Creek 49617.05
END DESCRIPTION:
XS GIS Cut Line= 3
      1536922.96      6843867.65      1537954.17      6843852.02
      1538735.41      6843596.82
#Sta/Elev= 30
  3967.9 1842.35    4350 1842.14    4500 1841.13    4540 1841.87    4570 1841.55
    4610 1840.11  4700.1 1839.62    4730 1839.72  4787.5 1836.83  4787.9 1836.33
  4792.1 1836.33  4792.5 1836.83    4810 1837.39    4870 1837.98  4890.1  1837.2
  4929.9 1836.85  4950.1 1837.66  5002.3 1837.05  5052.7 1837.89    5108 1837.69
  5250.5 1839.07  5294.7 1840.48  5389.3 1840.61  5510.8  1842.4  5568.2 1842.33
  5702.1 1843.98  5707.4  1843.6    5726 1843.94    5803 1843.63  5821.1 1844.01
#Mann= 5 ,-1 , 0
  3967.9    .045       0  4700.1     .07       0  4787.5     .07       0
  4792.5     .07       0    5108    .045       0
Bank Sta=4787.5,4792.5
XS Rating Curve= 0 ,0
Exp/Cntr=0.3,0.1

Type RM Length L Ch R = 1 ,49052   ,382,382,382
BEGIN DESCRIPTION:
Indian Creek 49267.05
END DESCRIPTION:
XS GIS Cut Line= 3
       1537663.5      6844661.24      1538205.17      6844296.66
      1538856.03      6843822.83
#Sta/Elev= 30
  4271.6 1838.12  4462.8 1838.14  4598.9 1836.54  4735.8 1836.36  4828.8 1834.89
  4927.5 1834.52  4936.8 1835.25  4966.2 1834.27  4973.8 1834.67  4984.5 1832.94
  4984.9 1832.44  4989.2 1832.44  4989.5 1832.94  5010.2 1833.81  5016.4 1833.25
  5045.8  1833.7  5051.9 1834.59  5109.9 1835.19  5131.5 1834.85  5182.4 1835.88
  5403.5 1839.57  5424.4 1840.06  5439.1 1841.27  5459.9 1840.69    5504 1841.42
  5524.8 1840.63    5531 1841.69    5575 1842.71    5640 1842.22  5729.6 1843.02
#Mann= 4 ,-1 , 0
  4271.6     .07       0  4984.5     .07       0  4989.5     .07       0
  5182.4    .045       0
Bank Sta=4984.5,4989.5
XS Rating Curve= 0 ,0
Exp/Cntr=0.3,0.1

Type RM Length L Ch R = 1 ,48670   ,61,61,61
BEGIN DESCRIPTION:
Indian Creek 48865.3
END DESCRIPTION:
XS GIS Cut Line= 3
      1538133.72      6844738.82      1538388.49      6844683.49
      1538938.56      6843805.12
#Sta/Elev= 30
  4548.1 1834.95  4673.5 1833.25  4733.6 1833.75  4816.4  1831.7  4868.3 1831.53
    4926 1832.03  4944.7 1831.46  4945.1 1830.96  4949.4 1830.96  4949.8 1831.46
  4968.7  1832.1  4977.9 1833.25  4999.1 1833.35    5005 1831.93  5014.4 1832.42
  5020.3 1833.54  5056.9 1833.28  5072.2 1833.94  5093.4 1833.54  5099.3 1834.12
  5151.2 1834.22  5229.7 1835.52  5324.5 1836.75  5397.5 1838.42  5470.6 1839.37
  5513.1  1840.6  5570.8 1840.75  5665.1 1842.62  5768.8 1842.64  5845.2 1844.01
#Mann= 4 ,-1 , 0
  4548.1     .07       0  4944.7     .07       0  4949.8     .07       0
  5229.7    .045       0
Bank Sta=4944.7,4949.8
XS Rating Curve= 0 ,0
Exp/Cntr=0.3,0.1

Type RM Length L Ch R = 1 ,48609   ,153,153,153
BEGIN DESCRIPTION:
Indian Creek 48593.65
END DESCRIPTION:
XS GIS Cut Line= 4
      1538172.05      6844752.16      1538488.97      6844730.63
      1538564.47      6844445.67       1539100.6      6843947.34
#Sta/Elev= 30
  4510.7 1834.27  4543.7 1833.63  4704.1 1832.86  4754.2 1831.76  4804.3 1831.34
  4862.1  1831.7  4874.5 1832.74  4909.6 1832.54  4944.6 1833.55  4955.2 1834.68
  4965.6 1834.83  4984.8  1833.2  4987.4 1831.05  4987.8 1830.55  4992.1 1830.55
  4992.5 1831.05  5006.9 1832.99    5025 1833.14  5030.2 1833.79  5048.3 1833.42
  5128.9 1833.82  5157.2 1834.57  5178.5 1834.38  5243.2 1835.42  5475.8 1839.32
  5532.5 1839.71  5553.5 1840.47  5652.7 1841.05  5723.5 1842.77  5855.1 1842.53
#Mann= 4 ,-1 , 0
  4510.7     .07       0  4987.4     .07       0  4992.5     .07       0
  5243.2    .045       0
Bank Sta=4987.4,4992.5
XS Rating Curve= 0 ,0
Exp/Cntr=0.3,0.1

Type RM Length L Ch R = 1 ,48456   ,165,165,165
BEGIN DESCRIPTION:
Indian Creek 16.0
END DESCRIPTION:
XS GIS Cut Line= 4
      1538292.79      6844771.33      1538556.96      6844764.36
      1538704.59      6844603.11      1538970.25      6844277.78
#Sta/Elev= 30
    4613 1833.45  4835.3 1831.62  4845.3 1832.44  4865.3 1837.49  4880.4 1839.93
  4908.8 1838.09  4929.8 1834.43  4951.3 1832.76  4958.1  1830.3  4965.5 1829.29
  4969.8 1826.53  4970.2 1826.03  4974.9 1826.53  4979.7 1827.63  4986.5  1826.7
  5000.7 1827.77  5014.9 1831.72    5029 1833.58  5064.2 1833.02  5085.8 1834.22
  5237.1 1835.66  5265.4  1835.9  5341.5  1837.4  5347.9 1838.85  5355.8 1837.98
  5370.2 1839.02    5391 1837.93  5440.5 1837.97  5476.9 1840.06  5515.9 1839.33
#Mann= 5 ,-1 , 0
    4613     .07       0  4969.8     .07       0  4974.9     .07       0
  5237.1    .045       0  5265.4     .07       0
Bank Sta=4969.8,4974.9
XS Rating Curve= 0 ,0
Exp/Cntr=0.3,0.1

Type RM Length L Ch R = 1 ,48291   ,105,105,105
BEGIN DESCRIPTION:
Indian Creek 14.0
END DESCRIPTION:
XS GIS Cut Line= 5
      1538295.92      6844792.06      1538628.43       6844839.6
       1538701.7      6844828.24      1538794.69      6844754.28
      1539019.81      6844682.95
#Sta/Elev= 30
  4633.9 1833.49  4862.8 1831.14  4863.2 1830.64  4867.9 1831.14    4922 1832.16
  4927.1  1831.6  4969.8 1833.27  4976.4 1834.75  4986.6 1835.12  5006.8 1835.26
  5017.4 1834.35  5048.1    1836  5053.4 1834.94  5067.9 1838.28  5074.3 1837.14
  5082.3 1838.15  5088.7 1836.46  5096.7 1837.37  5103.1 1835.56  5111.1 1836.43
  5117.5 1834.55  5131.9 1836.48  5138.3 1834.21  5146.4 1835.41  5152.7 1833.59
  5159.8 1832.89  5215.5  1835.2  5302.1 1834.32  5361.4 1837.24  5398.9 1836.02
#Mann= 3 ,-1 , 0
  4633.9     .07       0  4862.8     .07       0  4867.9     .07       0
Bank Sta=4862.8,4867.9
XS Rating Curve= 0 ,0
Exp/Cntr=0.3,0.1

Type RM Length L Ch R = 1 ,48186   ,53,53,53
BEGIN DESCRIPTION:
Indian Creek 48186.27
END DESCRIPTION:
XS GIS Cut Line= 3
       1538290.4      6844816.38      1538740.63      6844914.52
      1539241.89      6844952.51
#Sta/Elev= 30
  4551.8 1833.31  4740.7 1831.07  4802.1 1831.07  4812.4 1831.75  4832.8 1831.35
  4843.1 1831.94  4861.5 1831.07  4866.6 1831.43  4894.3 1827.97  4910.6 1826.89
  4951.9 1825.67  4952.3 1825.17  4956.7 1825.17  4957.1 1825.67  4959.6 1826.49
  4996.6 1825.96  5008.7 1827.21    5027 1827.81  5057.1 1831.23  5087.2 1831.68
  5107.2 1833.44  5137.3 1832.14  5207.5 1832.02  5254.9 1833.39  5307.8 1833.82
  5347.9 1835.49    5378  1834.6  5438.2  1834.1  5508.4 1835.44  5515.3 1836.18
#Mann= 3 ,-1 , 0
  4551.8     .07       0  4951.9     .07       0  4957.1     .07       0
Bank Sta=4951.9,4957.1
XS Rating Curve= 0 ,0
Exp/Cntr=0.3,0.1

Type RM Length L Ch R = 1 ,48133   ,106,106,106
BEGIN DESCRIPTION:
Indian Creek 13.0
END DESCRIPTION:
XS GIS Cut Line= 4
      1538267.97      6844892.87      1538659.31      6844953.46
      1538820.89      6844958.25      1539168.17      6845015.98
#Sta/Elev= 30
  4508.3 1833.39  4525.5 1832.73  4572.8 1833.46  4577.9 1832.79  4626.7 1832.89
  4667.2 1831.67  4766.9 1831.74  4796.1 1830.71  4796.5 1830.21  4800.9 1830.21
  4801.3 1830.71  4829.1 1831.14    4835 1832.44  4840.1 1831.13  4849.3 1831.56
  4879.7 1835.84  4898.1 1836.08  4902.8 1833.85    4910 1834.97    4930 1836.21
    5010 1835.34  5050.1 1831.07  5060.1 1831.24  5065.5 1832.81  5100.5 1831.26
    5151 1832.47    5283 1832.35    5354 1833.33  5394.5 1835.33    5418 1834.99
#Mann= 3 ,-1 , 0
  4508.3     .07       0  4796.1     .07       0  4801.3     .07       0
Bank Sta=4796.1,4801.3
XS Rating Curve= 0 ,0
Exp/Cntr=0.3,0.1

Type RM Length L Ch R = 1 ,48027   ,512,512,512
BEGIN DESCRIPTION:
Indian Creek 47903.49
END DESCRIPTION:
XS GIS Cut Line= 4
      1538248.32      6844962.38      1538639.68      6845022.98
      1538787.08      6845066.05      1539148.57       6845085.5
#Sta/Elev= 30
  4539.8 1833.43  4617.4 1832.09  4673.8 1832.06  4728.7 1830.41  4759.1 1831.08
  4779.3 1830.53  4819.8 1830.95  4829.9 1830.07    4840    1830  4850.1  1830.6
  4867.9 1830.79  4951.8 1829.22  4993.5 1829.62  5022.1 1828.67  5022.5 1828.17
  5026.9 1828.17  5027.3 1828.67  5041.6 1829.46  5046.8 1829.23  5075.1 1830.91
  5097.3 1830.27  5147.4 1829.89  5215.7 1830.72  5220.7 1830.38  5227.5 1830.84
  5257.5 1830.86  5317.6 1831.97  5377.7 1833.57  5417.8 1833.15  5451.4  1833.8
#Mann= 3 ,-1 , 0
  4539.8     .07       0  5022.1     .07       0  5027.3     .07       0
Bank Sta=5022.1,5027.3
XS Rating Curve= 0 ,0
Exp/Cntr=0.3,0.1

Type RM Length L Ch R = 1 ,47515   ,319,319,319
BEGIN DESCRIPTION:
Indian Creek 47515.24
END DESCRIPTION:
XS GIS Cut Line= 3
      1537740.65      6845633.27      1538693.75       6845523.9
      1539516.63      6845325.99
#Sta/Elev= 30
  4028.4 1833.75  4264.3 1833.78  4455.5 1831.43  4515.9 1831.78  4626.7 1830.03
  4707.2 1830.13  4821.6 1828.27  4878.3 1828.14  4898.4 1827.64  4928.6 1828.01
  4938.7 1827.02  4976.3 1825.55  4976.7 1825.05  4981.1 1825.05  4981.5 1825.55
  4992.9 1826.41  5009.6 1825.73    5061 1827.29  5076.9 1826.46    5133 1827.31
  5207.8 1827.24    5277 1827.84    5349    1829  5459.5 1828.88  5554.7  1830.9
  5626.7 1830.79  5688.4 1832.84  5758.3 1832.54  5822.1 1834.67  5834.1 1834.46
#Mann= 4 ,-1 , 0
  4028.4     .07       0  4976.3     .07       0  4981.5     .07       0
  5076.9    .045       0
Bank Sta=4976.3,4981.5
XS Rating Curve= 0 ,0
Exp/Cntr=0.3,0.1

Type RM Length L Ch R = 1 ,47196   ,499,499,499
BEGIN DESCRIPTION:
Indian Creek 47196.1
END DESCRIPTION:
XS GIS Cut Line= 3
      1537938.58      6846013.47      1538803.13      6845810.36
      1539469.84      6845450.96
#Sta/Elev= 30
  4109.8 1832.41  4136.9  1832.9  4286.3 1832.65  4371.1 1833.69  4376.3  1832.4
  4496.5  1830.1  4568.4 1830.14  4635.8 1828.48    4743 1827.47  4773.8 1828.42
  4845.7 1826.91  4927.9 1826.96  4948.5  1825.8  4985.4 1825.61  5012.6 1822.48
    5013 1821.98  5017.5 1821.98  5017.9 1822.48  5022.7 1823.22  5031.4 1826.08
  5037.1 1826.54  5045.5 1825.39  5094.1 1824.96  5295.4 1825.97  5452.4 1827.47
  5511.2 1828.74  5561.8 1828.69  5636.2  1830.6  5693.2  1830.6  5755.3 1832.45
#Mann= 4 ,-1 , 0
  4109.8     .07       0  5012.6     .07       0  5017.9     .07       0
  5094.1    .045       0
Bank Sta=5012.6,5017.9
XS Rating Curve= 0 ,0
Exp/Cntr=0.3,0.1

Type RM Length L Ch R = 1 ,46697   ,493,493,493
BEGIN DESCRIPTION:
Indian Creek 46696.85
END DESCRIPTION:
XS GIS Cut Line= 3
      1538277.11      6846706.18       1539032.3      6846169.73
      1539537.48      6845539.56
#Sta/Elev= 30
  4070.4 1831.55  4074.9 1832.33  4095.8 1832.05  4104.5  1831.2  4116.9    1831
  4325.4 1830.17  4505.4  1828.4  4555.9 1828.71  4591.5 1827.42  4619.8 1827.65
  4755.1 1825.57  4956.8 1823.95    5001 1823.11  5010.9 1822.46  5011.3 1821.96
  5015.9 1821.96  5016.4 1822.46    5036 1823.31  5106.4 1823.55  5178.4 1824.53
  5240.9 1824.24  5420.1 1825.38  5447.5 1826.12  5562.5 1827.45  5604.2 1828.71
  5653.8 1828.74  5701.7 1830.23  5717.8 1830.77  5767.9 1831.07  5804.4 1832.05
#Mann= 5 ,-1 , 0
  4070.4     .07       0  5010.9     .07       0  5016.4     .07       0
  5240.9    .045       0  5701.7     .07       0
Bank Sta=5010.9,5016.4
XS Rating Curve= 0 ,0
Exp/Cntr=0.3,0.1

Type RM Length L Ch R = 1 ,46204   ,475,475,475
BEGIN DESCRIPTION:
Indian Creek 46203.72
END DESCRIPTION:
XS GIS Cut Line= 3
      1538521.89      6846977.01      1539339.59      6846492.65
      1539943.77      6845753.04
#Sta/Elev= 30
  4035.5 1829.72  4182.6 1829.32  4336.6 1828.03  4364.5 1828.23  4468.5 1826.81
  4659.3 1824.98  4667.9 1824.92  4810.4 1822.98  4948.7    1822  5003.7 1820.44
  5004.2 1819.94  5009.4 1819.94  5009.9 1820.44  5029.1 1821.18  5101.1 1821.81
  5212.8 1822.39  5258.5 1823.24  5313.4 1823.91  5363.2 1823.86  5497.1 1825.11
  5568.2 1826.78  5624.9 1827.68  5661.6 1829.13  5703.2 1829.18  5725.4 1830.29
  5746.3 1830.69    5775 1830.45  5834.6 1831.52    5882 1832.79  5940.9 1832.65
#Mann= 12 ,-1 , 0
  4035.5     .07       0  4468.5    .045       0  4659.3     .07       0
  4667.9    .045       0  4810.4     .07       0  5003.7     .07       0
  5009.9     .07       0  5101.1    .045       0  5258.5     .07       0
  5363.2    .045       0  5568.2     .07       0  5834.6    .045       0
Bank Sta=5003.7,5009.9
XS Rating Curve= 0 ,0
Exp/Cntr=0.3,0.1

Type RM Length L Ch R = 1 ,45729   ,378,378,378
BEGIN DESCRIPTION:
Indian Creek 45728.78
END DESCRIPTION:
XS GIS Cut Line= 3
      1538600.01      6847424.94       1539532.3      6846872.86
      1540198.15      6845811.65
#Sta/Elev= 30
  3911.1  1828.4  4094.4 1828.01  4291.2 1827.53  4536.5 1825.42  4669.8 1824.03
  4860.5 1822.04  4902.5 1820.95  4934.6 1820.73  4956.1  1819.9  4971.7 1818.66
    4983  1818.6  4983.5  1818.1  4988.7  1818.1  4989.2  1818.6  5028.9 1819.68
  5260.4 1819.76  5348.2 1820.05  5413.5 1821.17  5487.6 1821.57  5588.5 1823.09
  5615.6 1824.27  5706.1 1824.86  5819.5 1826.62  5877.2 1827.94  5892.5 1828.82
  5956.6 1828.63  6023.3 1830.66    6081 1830.41  6175.3 1832.46  6247.4 1832.53
#Mann= 10 ,-1 , 0
  3911.1     .07       0  4094.4    .045       0  4536.5     .07       0
  4669.8    .045       0  4902.5     .07       0    4983     .07       0
  4989.2     .07       0  5260.4    .045       0  5487.6     .07       0
  5706.1    .045       0
Bank Sta=4983,4989.2
XS Rating Curve= 0 ,0
Exp/Cntr=0.3,0.1

Type RM Length L Ch R = 1 ,45351   ,406,406,406
BEGIN DESCRIPTION:
Indian Creek 45445.31
END DESCRIPTION:
XS GIS Cut Line= 3
      1539390.03      6847797.18      1539846.56      6847015.48
      1540212.44      6846259.18
#Sta/Elev= 30
  4058.2 1823.97  4280.1 1823.14  4318.2 1822.83  4485.7 1821.73  4535.9 1820.83
  4573.1 1821.05  4616.1 1820.35    4669 1820.39  4770.7 1819.09  4863.7 1818.55
  4888.1 1818.49  4915.4 1819.04  4937.4 1818.52  4968.8 1818.56  4991.4 1816.89
  5001.9 1816.57  5002.4 1816.07  5007.8 1816.07  5008.3 1816.57  5036.5 1817.87
  5153.1  1818.4  5426.1 1821.55  5567.8 1824.25  5595.4  1824.6    5618 1825.66
  5657.6 1825.53  5693.8 1825.93    5716 1826.81  5782.5 1827.14  5803.6  1827.4
#Mann= 9 ,-1 , 0
  4058.2    .045       0  4280.1     .07       0  4318.2    .045       0
  4863.7     .07       0  5001.9     .07       0  5008.3     .07       0
  5153.1    .045       0  5567.8     .07       0  5782.5    .045       0
Bank Sta=5001.9,5008.3
XS Rating Curve= 0 ,0
Exp/Cntr=0.3,0.1

Type RM Length L Ch R = 1 ,44945   ,170,170,170
BEGIN DESCRIPTION:
Indian Creek 45105.03
END DESCRIPTION:
XS GIS Cut Line= 3
      1539958.46      6848149.83      1540183.86       6847208.4
      1540389.33      6846341.46
#Sta/Elev= 30
    3998 1821.29  4046.9 1821.52  4061.6 1822.72  4082.1 1821.97  4088.9 1820.84
  4102.7 1821.79    4185 1820.08  4339.2  1819.9    4514 1817.76    4863  1816.6
  4863.5  1816.1  4869.4  1816.6    4915 1817.51  5007.6 1822.31  5034.6 1819.75
  5039.8 1822.44  5076.9 1819.17    5082 1821.25  5119.1 1819.65  5124.2 1821.65
  5202.8 1823.52  5208.7 1823.29  5213.8 1821.43  5250.9 1818.99  5472.4 1823.68
  5665.3 1825.51  5706.4 1827.38  5757.8  1826.9  5815.4 1828.35    5857 1828.04
#Mann= 3 ,-1 , 0
    3998    .035       0    4863    .035       0  4869.4    .035       0
Bank Sta=4863,4869.4
XS Rating Curve= 0 ,0
Exp/Cntr=0.3,0.1

Type RM Length L Ch R = 1 ,44775   ,341,341,341
BEGIN DESCRIPTION:
Indian Creek 44719.24
END DESCRIPTION:
XS GIS Cut Line= 3
      1539990.63      6848737.42      1540304.33      6847199.92
       1540600.6      6846357.89
#Sta/Elev= 30
  3546.8 1821.34  3556.4 1819.87  3566.6 1820.79  3678.9 1819.59  3801.4 1820.02
  4219.8 1819.26  4587.2 1817.15  4638.2  1816.3  4689.1 1816.39  4709.7 1817.68
  4744.8 1816.31  4992.3 1815.88  4997.4 1815.69  5002.4 1813.49  5002.9 1812.99
  5008.9 1813.49  5015.9 1815.15  5026.1 1815.83  5128.2 1816.79  5139.2 1817.42
  5226.4 1817.49  5468.8    1822  5525.4 1824.68  5556.4 1823.79  5595.1 1824.58
  5626.9 1826.14  5731.6 1826.17  5785.9 1827.79  5886.4 1827.88  6008.6 1829.71
#Mann= 3 ,-1 , 0
  3546.8     .07       0  5002.4     .07       0  5008.9     .07       0
Bank Sta=5002.4,5008.9
XS Rating Curve= 0 ,0
Exp/Cntr=0.3,0.1

Type RM Length L Ch R = 1 ,44434   ,483,483,483
BEGIN DESCRIPTION:
Indian Creek 44195.32
END DESCRIPTION:
XS GIS Cut Line= 3
      1540042.72      6848753.06      1540597.45      6847396.86
      1540904.61      6846862.98
#Sta/Elev= 30
  3598.5 1821.53  3613.6 1819.95  4425.1 1817.43  4438.9 1816.66  4754.1 1814.13
  4778.1 1815.11  4846.5 1813.57  4868.1 1810.35  4878.9 1810.76  4884.9 1812.37
    4887  1810.1  4887.5  1809.6  4893.6  1810.1  4908.9 1813.42  4914.3  1812.8
  4938.4 1814.12  4986.4 1813.94  4997.7 1811.96  5021.2 1814.22  5030.1 1813.11
  5039.8 1813.51  5045.2 1812.82  5068.5  1814.2  5154.8 1816.08  5192.2 1818.02
    5208 1817.17  5294.2 1819.73  5523.9 1824.43  5594.6 1824.23  5679.7 1825.61
#Mann= 3 ,-1 , 0
  3598.5     .07       0    4887     .07       0  4893.6     .07       0
Bank Sta=4887,4893.6
XS Rating Curve= 0 ,0
Exp/Cntr=0.3,0.1

Type RM Length L Ch R = 1 ,43951   ,326,326,326
BEGIN DESCRIPTION:
Indian Creek 43951.44
END DESCRIPTION:
XS GIS Cut Line= 3
      1540209.38      6848794.74      1540714.59      6847893.69
      1541516.65      6847086.41
#Sta/Elev= 30
    3969  1820.7  3986.6 1819.48  4057.4 1818.78  4235.4 1818.36  4779.2 1813.67
    4814 1814.47  4859.5 1813.35  4916.8 1813.22  4954.3 1814.61  4970.3 1812.99
    4976    1811  4988.7 1810.34  4989.2 1809.84  4995.3 1810.34  4997.3 1811.83
  5034.6 1813.07  5048.8 1812.39  5211.4 1813.36  5381.1 1818.38  5430.6 1819.17
  5550.8 1818.71  5586.2 1819.38  5593.2 1818.47  5607.4 1818.44  5678.1 1821.23
    5869 1821.68  5982.2 1823.31  6017.5 1824.61  6088.2 1824.21    6140 1824.96
#Mann= 3 ,-1 , 0
    3969     .07       0  4988.7     .07       0  4995.3     .07       0
Bank Sta=4988.7,4995.3
XS Rating Curve= 0 ,0
Exp/Cntr=0.3,0.1

Type RM Length L Ch R = 1 ,43625   ,630,630,630
BEGIN DESCRIPTION:
Indian Creek 43625.381
END DESCRIPTION:
XS GIS Cut Line= 3
      1540297.91      6848846.83      1541047.92       6847961.4
      1541661.05      6847493.76
#Sta/Elev= 30
  3982.3 1819.39  4021.6 1820.21  4035.8 1818.89  4589.5 1813.26  4767.1 1811.97
  4909.3 1812.51  4998.2 1810.25  4998.7 1809.75  5004.8 1810.25  5008.1 1811.48
  5207.1 1814.88  5300.6 1814.54  5342.2 1815.63  5350.5 1814.34  5356.8 1816.36
    5365 1814.86  5371.3 1816.97  5385.8 1812.74  5392.1 1814.37  5400.4 1813.71
  5406.6  1815.8  5570.8 1820.15  5692.4 1820.74    5706 1822.85  5742.7 1824.26
  5749.6 1822.76  5755.9 1824.12  5834.8 1822.88  5870.2 1824.04  5913.8 1822.77
#Mann= 3 ,-1 , 0
  3982.3     .07       0  4998.2     .07       0  5004.8     .07       0
Bank Sta=4998.2,5004.8
XS Rating Curve= 0 ,0
Exp/Cntr=0.3,0.1

Type RM Length L Ch R = 1 ,42995   ,432,432,432
BEGIN DESCRIPTION:
Indian Creek 42995
END DESCRIPTION:
XS GIS Cut Line= 3
      1540381.26      6848961.39      1541131.25      6848570.77
      1541989.53       6847712.5
#Sta/Elev= 30
  4150.4 1818.83  4214.2 1818.15  4280.5 1818.76  4319.1 1817.79  4324.7 1818.87
  4341.2 1819.04  4413.9 1816.73  4490.3 1815.71  4926.6 1810.86  4948.7 1811.46
  4965.2 1810.48  4974.3 1807.43  4974.8 1806.93  4981.1 1807.43  4992.9 1809.16
  5078.4 1809.17  5127.9 1808.23  5212.8 1810.65    5234 1809.65  5297.6 1809.19
  5424.9 1811.63  5460.2 1813.54  5488.5 1814.35  5495.6  1813.8  5502.7 1815.02
  5516.8 1815.38  5559.2  1816.1  5622.9 1815.75  5912.8 1819.92  6209.8  1820.5
#Mann= 3 ,-1 , 0
  4150.4     .07       0  4974.3     .07       0  4981.1     .07       0
Bank Sta=4974.3,4981.1
XS Rating Curve= 0 ,0
Exp/Cntr=0.3,0.1

Type RM Length L Ch R = 1 ,42563   ,180,180,180
BEGIN DESCRIPTION:
Indian Creek 42562.69
END DESCRIPTION:
XS GIS Cut Line= 3
      1540553.11      6849086.41      1541521.88      6848602.02
      1542224.55      6847852.51
#Sta/Elev= 30
  3919.4 1818.21  3999.8 1817.11  4083.6 1817.34  4122.7 1816.24  4240.1 1816.47
  4262.5 1815.32  4379.9  1813.7  4569.9 1811.29    4693 1810.81  4804.8 1808.78
  4871.8 1809.39  4955.6 1807.89  4972.4  1807.1    4980 1805.74  4980.5 1805.24
  4987.3 1805.74  5035.7 1806.81    5064 1808.05  5071.3 1809.19  5134.8 1808.83
  5241.1  1810.6  5382.4 1815.96  5446.4 1815.48  5613.3 1817.82  5729.2 1819.58
  5792.3 1819.26  5835.6 1819.62  5911.6 1819.79  5999.4 1819.68  6029.9 1819.82
#Mann= 8 ,-1 , 0
  3919.4     .07       0    4980     .07       0  4987.3     .07       0
  5613.3    .035       0  5792.3     .07       0  5835.6    .035       0
  5911.6     .07       0  5999.4    .035       0
Bank Sta=4980,4987.3
XS Rating Curve= 0 ,0
Exp/Cntr=0.3,0.1

Type RM Length L Ch R = 1 ,42383   ,368,368,368
BEGIN DESCRIPTION:
Indian Creek 42383.28
END DESCRIPTION:
XS GIS Cut Line= 3
      1540803.13      6849195.77      1541672.92      6848669.73
      1542360.23      6847883.49
#Sta/Elev= 30
  3974.6 1816.24    4024 1816.42  4097.7 1815.11  4156.7 1815.46  4246.6 1813.56
  4303.3 1813.91  4309.2 1813.06  4330.5  1814.2    4346 1813.83  4351.9 1812.68
  4419.7 1811.75  4788.4 1808.08  4843.5 1808.02  4935.1 1807.59  4958.5 1806.29
  5015.2 1806.06  5025.7    1805  5026.2  1804.5  5033.1    1805  5043.7  1807.5
  5057.9 1808.93  5142.4 1809.11  5185.1 1810.08  5213.6 1812.22    5242 1812.33
  5262.9 1813.46  5284.7 1815.51  5580.4 1817.61  5687.1 1818.89  6035.4 1819.72
#Mann= 9 ,-1 , 0
  3974.6     .07       0  4156.7    .045       0  4246.6     .07       0
  4788.4    .035       0  4843.5     .07       0  5025.7     .07       0
  5033.1     .07       0  5580.4    .035       0  5687.1     .07       0
Bank Sta=5025.7,5033.1
XS Rating Curve= 0 ,0
Exp/Cntr=0.3,0.1

Type RM Length L Ch R = 1 ,42015   ,405,405,405
BEGIN DESCRIPTION:
Indian Creek 41979
END DESCRIPTION:
XS GIS Cut Line= 3
       1541394.2      6849256.35      1541698.84      6848975.27
      1542324.61      6848382.43
#Sta/Elev= 30
  4625.6 1809.53  4768.2 1808.77  4816.3 1808.61  4823.1 1809.47  4844.4  1809.7
  4872.4    1808  4922.3 1808.07  4930.8 1807.48  4936.5 1806.72  4979.1 1807.26
  4996.3  1804.4  4996.8  1803.9  5003.3  1803.9  5003.8  1804.4  5014.2 1805.18
  5056.7 1805.16  5099.2  1806.2  5184.1 1806.16  5198.3 1806.31  5205.2  1807.3
  5240.8 1806.79  5346.7 1808.02  5488.3 1810.03  5665.5 1813.56  5778.4 1815.82
  5799.4 1816.84  5806.3 1817.85  5812.4 1817.65  5848.8 1817.06  5902.1 1817.58
#Mann= 7 ,-1 , 0
  4625.6    .045       0  4768.2     .07       0  4930.8    .035       0
  4996.3    .035       0  5003.8    .035       0  5665.5     .07       0
  5812.4    .035       0
Bank Sta=4996.3,5003.8
XS Rating Curve= 0 ,0
Exp/Cntr=0.3,0.1

Type RM Length L Ch R = 1 ,41610   ,566,566,566
BEGIN DESCRIPTION:
Indian Creek 12.0
END DESCRIPTION:
XS GIS Cut Line= 5
      1541605.11      6849234.18      1541988.76      6849108.32
      1542094.38      6849117.74      1542144.31      6849077.42
      1542332.85      6848416.79
#Sta/Elev= 30
  4645.7 1808.17  4741.7 1807.45  4846.4 1807.41  5028.3 1804.65  5028.8 1804.15
  5035.9 1804.65  5037.3 1805.92  5065.8 1809.22  5095.9 1809.84  5101.5 1809.54
  5106.6 1806.94  5146.1 1809.31  5183.7 1808.58  5191.7 1809.59  5198.1 1808.14
  5206.1 1809.43  5212.5  1807.7    5222 1809.25  5315.6 1806.96  5395.9 1808.21
  5416.7 1810.11  5447.8  1809.9  5525.7 1810.38  5562.3 1812.73  5628.6 1813.15
  5714.9 1814.68  5776.4 1815.43  5832.6 1816.45  5864.5 1818.59  5906.7 1817.28
#Mann= 9 ,-1 , 0
  4645.7    .045       0  4741.7     .07       0  5028.3     .07       0
  5035.9     .07       0  5447.8    .035       0  5525.7     .07       0
  5628.6    .035       0  5714.9     .07       0  5776.4    .035       0
Bank Sta=5028.3,5035.9
XS Rating Curve= 0 ,0
Exp/Cntr=0.3,0.1

Type RM Length L Ch R = 1 ,41044   ,190,190,190
BEGIN DESCRIPTION:
Indian Creek 41216.83
END DESCRIPTION:
XS GIS Cut Line= 4
      1541991.26      6849303.85      1542272.41      6849251.68
      1542746.89      6849343.79      1543202.78      6849021.32
#Sta/Elev= 30
  4576.7 1805.78  4627.7  1805.5  4733.1 1805.26  4747.1 1804.38  4794.1 1804.89
  4834.8 1803.37  4916.2 1803.12  4948.4 1802.11  5004.1 1800.72  5004.6 1800.22
  5011.7 1800.72  5025.1 1802.85  5038.5  1803.4  5048.6 1802.73  5099.6 1803.19
  5150.5 1802.27  5221.8 1803.51  5293.8 1802.68  5340.4 1803.99  5363.4 1803.68
  5369.5 1804.38  5378.1 1803.69  5413.8 1803.77  5527.4 1806.32  5571.4 1808.13
  5592.3 1807.87    5708 1810.39  5764.6  1810.4  5779.4 1811.27  5904.4 1811.21
#Mann= 5 ,-1 , 0
  4576.7     .07       0  4627.7    .035       0  4948.4     .07       0
  5004.1     .07       0  5011.7     .07       0
Bank Sta=5004.1,5011.7
XS Rating Curve= 0 ,0
Exp/Cntr=0.3,0.1

Type RM Length L Ch R = 1 ,40854   ,479,479,479
BEGIN DESCRIPTION:
Indian Creek 40844.5
END DESCRIPTION:
XS GIS Cut Line= 3
       1541951.3      6849390.96      1542674.26      6849443.78
      1543145.35      6849541.48
#Sta/Elev= 30
  4440.5 1806.17  4544.5 1805.02  4674.8 1804.72  4889.2 1803.28  4905.4 1803.39
  4955.6  1800.6  4975.6 1801.06  5081.6 1799.76  5082.1 1799.26  5089.7 1799.26
  5090.2 1799.76  5129.1 1800.45  5146.1 1801.05  5152.9 1801.87  5157.9 1801.36
  5168.3 1801.59  5176.4 1802.91  5186.6 1803.08  5196.8 1801.87  5211.4 1802.03
  5227.4 1801.43  5256.5 1802.18  5311.8 1802.36  5421.5 1804.22    5452 1805.37
  5457.1 1804.61    5493 1806.13  5507.3 1805.96  5523.6 1807.02  5646.5 1808.42
#Mann= 5 ,-1 , 0
  4440.5    .035       0  4889.2     .07       0  5081.6     .07       0
  5090.2     .07       0  5129.1    .035       0
Bank Sta=5081.6,5090.2
XS Rating Curve= 0 ,0
Exp/Cntr=0.3,0.1

Type RM Length L Ch R = 1 ,40375   ,538,538,538
BEGIN DESCRIPTION:
Indian Creek 39957.473
END DESCRIPTION:
XS GIS Cut Line= 3
      1541823.55      6849953.63      1542755.91      6849847.87
      1543500.27      6849751.54
#Sta/Elev= 30
  4162.7 1807.45  4405.7 1804.88  4527.3 1804.46  4596.9 1803.26  4687.5 1803.43
  4928.4 1800.55  5009.5  1799.2  5055.2 1799.39  5090.1 1800.53  5103.1 1799.46
  5110.2 1797.56  5120.3  1797.1  5137.2 1798.97  5190.9 1801.05    5211 1800.44
  5231.2  1797.4  5261.5 1795.07  5277.3 1794.71  5277.8 1794.21    5286 1794.71
  5301.8 1797.53    5370 1802.37  5392.5 1804.89  5402.6 1804.53  5463.1 1807.44
  5584.1 1809.17  5594.2 1810.22  5654.7 1809.84    5695 1810.82  5851.6 1812.07
#Mann= 4 ,-1 , 0
  4162.7    .045       0  4928.4     .07       0  5277.3     .07       0
    5286     .07       0
Bank Sta=5277.3,5286
XS Rating Curve= 0 ,0
Exp/Cntr=0.3,0.1

Type RM Length L Ch R = 1 ,39837   ,503,503,503
BEGIN DESCRIPTION:
Indian Creek 39837
END DESCRIPTION:
XS GIS Cut Line= 3
      1541678.15      6850315.57      1542756.25       6850336.4
      1543725.03      6850200.98
#Sta/Elev= 30
  3917.5 1808.86  3964.4 1808.01  4014.4 1808.31  4084.4 1806.71  4144.4 1806.79
  4224.4  1805.2  4504.5  1803.3  4574.5 1801.82  4624.5 1801.94  4684.5 1800.25
  4764.5 1800.37  4834.5 1799.06  4904.5 1799.48  4924.5 1797.37  4976.7 1796.79
  5065.2 1797.41  5070.9  1796.5  5071.4    1796  5079.7  1796.5  5119.8 1797.21
  5190.9 1798.67  5288.5 1800.55    5425 1803.44  5479.2 1804.98  5519.6 1804.91
    5611  1806.9  5744.7 1808.41  5761.9 1807.63  5811.7 1808.39    5974 1809.19
#Mann= 10 ,-1 , 0
  3917.5    .045       0  4976.7     .07       0  5070.9     .07       0
  5079.7     .07       0  5119.8    .035       0  5190.9     .07       0
  5288.5    .035       0    5425     .07       0    5611    .035       0
  5811.7    .045       0
Bank Sta=5070.9,5079.7
XS Rating Curve= 0 ,0
Exp/Cntr=0.3,0.1

Type RM Length L Ch R = 1 ,39334   ,417,417,417
BEGIN DESCRIPTION:
Indian Creek 39570.07
END DESCRIPTION:
XS GIS Cut Line= 4
      1542117.84      6850670.04      1542873.24      6850732.83
      1542991.03      6850758.98      1543799.94      6850426.34
#Sta/Elev= 30
  4159.9 1803.63  4237.3 1803.55  4314.5 1801.99  4598.6 1800.11  4698.9 1798.03
  4739.1 1798.52  4759.1 1796.34  4802.5 1795.47  4824.9 1794.82  4825.4 1794.32
  4833.9 1794.82  4849.4 1796.28  4879.5    1797  4899.6 1797.06  4916.3 1795.74
  4921.8 1797.42  4960.2 1796.13  4965.3 1797.24  5008.9 1795.57    5014 1796.51
  5032.4 1796.74  5187.3 1795.93  5295.9 1797.76  5317.9 1798.57  5432.1 1799.52
  5517.8 1801.69  5608.5 1804.45  5649.2 1804.81    5670  1805.7  5913.2 1807.67
#Mann= 7 ,-1 , 0
  4159.9    .045       0  4802.5     .07       0  4824.9     .07       0
  4833.9     .07       0  5295.9    .035       0  5517.8     .07       0
  5649.2    .045       0
Bank Sta=4824.9,4833.9
XS Rating Curve= 0 ,0
Exp/Cntr=0.3,0.1

Type RM Length L Ch R = 1 ,38917   ,366,366,366
BEGIN DESCRIPTION:
Indian Creek 39234.33
END DESCRIPTION:
XS GIS Cut Line= 6
      1542402.39      6851099.16       1542979.2      6850993.59
      1543197.04      6851019.46      1543252.59      6851001.42
       1543260.3       6850918.2      1544091.86      6850658.52
#Sta/Elev= 30
  4162.7 1801.81  4515.5 1798.43  4592.3 1797.51  4622.8 1798.16    4633 1799.55
  4639.7 1797.99  4663.5 1797.02  4717.8 1798.03  4749.1 1797.55  4754.9 1796.71
  4824.6 1798.22  4829.7 1796.51  4835.5 1796.54  4885.8 1800.29    4906 1800.64
  4976.8 1799.08  5019.2 1799.08  5115.5 1799.17  5136.3 1795.47  5188.7 1795.47
    5190  1794.9  5190.5  1794.4    5199  1794.9  5201.8 1795.26  5226.9 1795.84
  5232.2 1795.29  5272.4 1796.84  5306.4  1797.3  5691.6 1803.99  5981.6 1805.77
#Mann= 9 ,-1 , 0
  4162.7    .045       0  4515.5     .07       0  4717.8     .16       0
  5019.2     .07       0    5190     .07       0    5199     .07       0
  5201.8    .035       0  5272.4     .07       0  5306.4    .045       0
Bank Sta=5190,5199
XS Rating Curve= 0 ,0
Exp/Cntr=0.3,0.1

Type RM Length L Ch R = 1 ,38551   ,238,238,238
BEGIN DESCRIPTION:
Indian Creek 38551.37
END DESCRIPTION:
XS GIS Cut Line= 5
      1542178.48      6851295.08      1543138.52      6851337.69
      1543261.46      6851367.65      1543340.27      6851385.71
      1544086.59      6851270.03
#Sta/Elev= 30
  3918.6  1802.9  4385.6 1800.44  4535.7 1799.22  4625.8  1797.6  4675.9 1798.48
  4695.9 1796.63  4859.3 1794.43  4927.4 1794.01  4943.6 1790.01  4948.7 1790.06
  4958.3 1787.29  4978.9 1785.53  5036.5 1784.68  5045.1 1785.18  5050.8 1787.45
  5070.5 1792.27  5081.6 1793.44    5112  1794.1  5122.1 1792.31  5142.4 1793.88
    5197 1793.66  5263.8 1793.43  5294.1 1794.26  5354.9 1794.19  5493.9 1795.96
    5537 1795.55  5659.8 1797.19  5697.6 1798.02    5819 1799.09  5842.2 1800.33
#Mann= 7 ,-1 , 0
  3918.6    .045       0  4859.3     .07       0  4978.9     .04       0
  5045.1     .07       0    5197    .035       0  5659.8    .063       0
  5697.6    .035       0
Bank Sta=4978.9,5045.1
XS Rating Curve= 0 ,0
Exp/Cntr=0.3,0.1

Type RM Length L Ch R = 1 ,38313   ,200,200,200
BEGIN DESCRIPTION:
Indian Creek 10.0
END DESCRIPTION:
XS GIS Cut Line= 5
      1542156.27      6851515.91       1543136.7      6851567.39
      1543275.17      6851603.66      1543342.28      6851571.62
      1544177.59      6851460.24
#Sta/Elev= 30
  3841.8 1802.93  4341.2 1800.79  4501.4 1798.64  4611.6 1798.16  4631.6 1796.85
  4691.7 1795.78  4837.8  1794.5  4863.2 1794.24  4873.5  1795.2  4935.5 1795.51
  4965.4 1793.36  5053.9 1793.22  5059.5 1791.22    5060 1790.72  5068.6 1791.22
  5084.2 1793.15  5144.7 1792.22  5225.4 1792.85  5316.2 1792.44  5346.5 1793.34
  5376.8 1792.94  5437.1 1793.72  5467.6 1793.76  5488.7 1794.93  5548.3 1794.18
  5689.7 1796.22  5760.1 1797.49  5780.3 1796.87  5859.4 1798.95  5883.8 1798.69
#Mann= 6 ,-1 , 0
  3841.8    .045       0  4837.8     .07       0  5059.5     .07       0
  5068.6     .07       0  5437.1    .035       0  5689.7    .063       0
Bank Sta=5059.5,5068.6
XS Rating Curve= 0 ,0
Exp/Cntr=0.3,0.1

Type RM Length L Ch R = 1 ,38113   ,302,302,302
BEGIN DESCRIPTION:
Indian Creek 38112.6
END DESCRIPTION:
XS GIS Cut Line= 3
      1542167.71      6851716.61      1543303.13      6851789.52
      1544547.96      6851784.31
#Sta/Elev= 30
  3860.2 1802.27  4188.2    1801  4258.3 1801.85  4298.4 1800.29  4639.1 1797.71
  4659.1 1798.16  4709.2 1796.15  4819.5 1794.48  4859.5 1795.08  4873.9  1794.4
  4895.4 1792.83  4939.7 1793.07  4959.8  1791.7  4969.8 1790.23  4985.2 1789.58
  4985.7 1789.08  4994.5 1789.58  5049.8 1789.78  5059.8 1791.39  5069.8 1791.69
  5179.8 1790.68  5289.8 1790.82  5499.8 1792.09  5559.8  1793.3  5679.8 1793.63
  5719.8 1794.59  5879.8 1794.62  5919.8 1795.99    5980 1796.55  6242.8 1798.58
#Mann= 5 ,-1 , 0
  3860.2    .045       0  4873.9     .07       0  4985.2     .07       0
  4994.5     .07       0    5980    .035       0
Bank Sta=4985.2,4994.5
XS Rating Curve= 0 ,0
Exp/Cntr=0.3,0.1

Type RM Length L Ch R = 1 ,37811   ,298,298,298
BEGIN DESCRIPTION:
Indian Creek 37810.92
END DESCRIPTION:
XS GIS Cut Line= 3
      1542318.72      6852128.07      1543297.92      6852091.61
      1544589.59      6852018.69
#Sta/Elev= 30
  4012.9 1801.13  4016.9 1801.19    4247  1800.7  4279.4 1801.55  4319.4 1799.53
  4629.6 1797.49  4669.6 1798.33  4729.7 1795.48  4818.9 1795.14  4899.8 1793.46
  4955.1 1793.46  4969.8  1792.5  4988.8 1789.09  5014.9 1788.18  5015.4 1787.68
    5025 1788.18    5060 1788.41    5080 1790.84  5240.3 1789.96  5380.5 1790.12
    5711 1792.49  5821.2 1792.17    5912 1793.16  6011.5  1795.7  6029.6 1794.93
  6061.6 1795.67  6081.6 1795.16  6141.7 1797.07  6201.8 1796.85  6286.5 1795.35
#Mann= 7 ,-1 , 0
  4012.9     .07       0  4016.9    .035       0    4247    .045       0
  4818.9     .07       0  5014.9     .07       0    5025     .07       0
    5912    .035       0
Bank Sta=5014.9,5025
XS Rating Curve= 0 ,0
Exp/Cntr=0.3,0.1

Type RM Length L Ch R = 1 ,37513   ,228,228,228
BEGIN DESCRIPTION:
Indian Creek 37512.54
END DESCRIPTION:
XS GIS Cut Line= 3
      1542459.41      6852430.15      1543292.71      6852388.48
      1544880.66      6852419.72
#Sta/Elev= 30
  4148.4 1801.63  4254.1 1801.52  4485.9 1798.63  4502.2 1798.73  4592.6 1798.66
    4690 1797.51  4884.9 1794.39  4904.9 1793.26  4927.4 1790.26    4945 1789.87
    4955  1790.9  4986.4 1788.09    4990 1786.02  4990.5 1785.52  5000.1 1786.02
    5035  1788.1  5121.8 1788.65  5185.1 1789.24  5211.3 1787.69  5345.1 1789.77
  5385.1 1788.84  5506.7 1789.96    5886  1790.2  5975.2 1791.72  5996.3 1791.03
  6195.3 1791.65  6215.3 1792.51  6275.3 1791.31  6355.3 1792.11    6571 1791.46
#Mann= 12 ,-1 , 0
  4148.4     .07       0  4485.9    .035       0  4502.2     .07       0
  4592.6    .035       0    4690     .07       0  4927.4    .035       0
    4990    .035       0  5000.1    .035       0  5121.8     .07       0
  5506.7    .035       0    5886    .063       0  5996.3    .094       0
Bank Sta=4990,5000.1
XS Rating Curve= 0 ,0
Exp/Cntr=0.3,0.1

Type RM Length L Ch R = 1 ,37285   ,358,358,358
BEGIN DESCRIPTION:
Indian Creek 37284.71
END DESCRIPTION:
XS GIS Cut Line= 3
       1542438.6       6852456.2       1543407.3      6852581.19
      1544589.62      6852591.61
#Sta/Elev= 30
  4026.7 1801.53  4194.5 1801.28  4236.4 1800.03  4325.6 1799.49  4398.3 1798.06
  4426.4 1798.81  4456.6 1797.84  4497.7  1797.8  4539.1 1797.66  4658.3 1796.13
  4678.5 1796.53  4819.6 1793.43  4839.8 1793.57  4858.1 1792.15  4942.5 1789.93
    4991 1787.26  4994.7 1786.38  4995.2 1785.88  5004.9 1786.38  5041.1 1786.42
  5061.1 1787.12  5071.1 1788.31  5144.6 1787.68  5271.1 1788.79  5521.2 1788.82
  5551.2 1790.06  5786.9 1789.49  5881.2 1790.57  5941.8 1790.39  6185.8 1791.99
#Mann= 10 ,-1 , 0
  4026.7    .063       0  4236.4     .07       0  4398.3    .035       0
  4497.7     .07       0  4539.1    .035       0  4994.7    .035       0
  5004.9    .035       0  5144.6     .07       0  5786.9    .063       0
  5941.8    .094       0
Bank Sta=4994.7,5004.9
XS Rating Curve= 0 ,0
Exp/Cntr=0.3,0.1

Type RM Length L Ch R = 1 ,36927   ,426,426,426
BEGIN DESCRIPTION:
Indian Creek 36927.49
END DESCRIPTION:
XS GIS Cut Line= 3
      1542568.72      6853003.07      1543386.46      6852935.36
      1544667.68      6853122.85
#Sta/Elev= 30
  4161.4 1798.52  4283.2 1797.38  4378.4 1797.58  4488.3 1795.98  4779.8 1791.52
    4830 1791.65    4840 1791.41  4860.1 1788.86  4940.3 1787.32  4970.4 1785.67
  4973.5 1784.88    4974 1784.38  4983.8 1784.88  4990.6 1786.01  5035.4 1786.21
  5051.2 1788.38  5105.3 1787.36  5111.8 1788.39  5170.1 1789.65  5192.7 1788.72
  5202.8 1789.55  5212.9 1788.68  5273.5    1788  5309.9 1786.13  5344.3  1785.8
  5404.9 1786.89  5819.3 1787.74  5869.8 1787.16  5980.9 1787.98  6276.8  1787.9
#Mann= 5 ,-1 , 0
  4161.4    .045       0  4488.3    .035       0  4973.5    .035       0
  4983.8    .035       0  5980.9    .094       0
#XS Ineff= 2 , 0
       0                    5550       0    1789
Permanent Ineff=
       F       F
Bank Sta=4973.5,4983.8
XS Rating Curve= 0 ,0
Exp/Cntr=0.3,0.1

Type RM Length L Ch R = 1 ,36501   ,243,243,243
BEGIN DESCRIPTION:
Indian Creek 36500.83
END DESCRIPTION:
XS GIS Cut Line= 3
      1542396.91      6853310.35      1543709.38      6853200.98
      1544651.03      6853148.96
#Sta/Elev= 30
  3688.4 1797.33  3907.2 1795.93  4208.3 1795.24  4368.8 1793.39  4478.5 1791.11
  4519.4 1791.53  4579.6 1789.24  4659.8 1788.46  4737.7 1786.43  4840.5 1786.38
  4934.7 1785.18  4970.9 1784.98  4985.8 1781.64  4986.3 1781.14  4996.1 1781.64
  5000.7 1783.23  5005.4 1783.23    5011 1785.05  5091.2 1783.53  5148.2 1783.48
  5171.3 1783.66  5181.3 1784.72  5221.4 1785.89    5334 1786.26  5391.6 1785.63
    5568 1786.65    5632 1786.51  5697.8 1787.71  5852.3 1788.52  5948.5 1787.49
#Mann= 7 ,-1 , 0
  3688.4    .045       0  4478.5     .07       0  4934.7    .035       0
  4985.8    .035       0  4996.1    .035       0    5568     .07       0
  5697.8    .094       0
Bank Sta=4985.8,4996.1
XS Rating Curve= 0 ,0
Exp/Cntr=0.3,0.1
