HEC-RAS study Little Elm Creek 2.prj: Little Elm Creek 2 Base Level Engineering

--- Little Elm Creek 2.g01 (geometry) --- (continued)

Type RM Length L Ch R = 1,25969,226,226,226
BEGIN DESCRIPTION:
Little Elm Creek 2 25969.25
END DESCRIPTION:
XS GIS Cut Line= 3
      1498503.43      6763135.02      1498636.23      6762885.04
      1498740.21      6762479.53
#Sta/Elev= 30
  4721.0 2360.18  4762.9 2357.95  4795.1 2358.13  4813.8 2356.65  4844.7 2355.40
  4883.0 2352.43  4898.8 2350.34  4932.8 2342.06  4943.3 2340.29  4965.3 2333.00
  4970.9 2330.57  4978.1 2324.94  4987.3 2319.62  4996.4 2316.32  4996.9 2315.82
  5002.7 2316.32  5032.0 2320.30  5063.8 2321.54  5093.9 2321.61  5175.8 2327.19
  5216.6 2336.67  5221.8 2336.96  5228.1 2338.97  5257.4 2345.12  5262.5 2345.08
  5279.7 2348.96  5298.1 2351.58  5338.9 2354.43  5420.5 2356.74  5422.7 2356.28
#Mann=4,-1,0
  4721.0    0.07       0  4813.8    0.16       0  4996.4    0.07       0
  5002.7    0.16       0
Bank Sta=4996.4,5002.7
Exp/Cntr=0.3,0.1

Type RM Length L Ch R = 1,25743,172,172,172
BEGIN DESCRIPTION:
Little Elm Creek 2 25742.77
END DESCRIPTION:
XS GIS Cut Line= 3
      1498578.92      6763179.33      1498839.36      6762965.77
      1499052.90      6762679.31
#Sta/Elev= 30
  4668.1 2358.35  4683.2 2357.03  4737.7 2353.38  4772.8 2352.23  4787.2 2349.81
  4793.6 2349.64  4865.4 2336.13  4900.6 2327.96  4935.7 2323.29  4972.3 2321.28
  4978.8 2318.36  4993.1 2316.73  4999.2 2315.16  5004.9 2315.16  5011.3 2312.86
  5011.8 2312.36  5017.8 2312.86  5036.4 2318.10  5078.0 2319.16  5114.4 2322.89
  5136.5 2327.68  5142.7 2330.05  5151.1 2330.88  5164.3 2336.03  5192.7 2343.88
  5242.8 2354.73  5251.1 2354.47  5286.6 2357.54  5338.0 2358.77  5362.2 2359.55
#Mann=5,-1,0
  4668.1    0.07       0  4683.2    0.16       0  5011.3    0.07       0
  5017.8    0.16       0  5338.0    0.07       0
Bank Sta=5011.3,5017.8
Exp/Cntr=0.3,0.1

Type RM Length L Ch R = 1,25571,148,148,148
BEGIN DESCRIPTION:
Little Elm Creek 2 25571.4
END DESCRIPTION:
XS GIS Cut Line= 3
      1498599.80      6763275.64      1498993.01      6763020.45
      1499162.29      6762812.11
#Sta/Elev= 30
  4534.8 2358.83  4564.0 2357.00  4600.7 2355.60  4636.9 2351.91  4673.2 2349.72
  4688.3 2346.71  4696.0 2343.92  4718.6 2340.12  4724.6 2340.45  4754.9 2336.09
  4760.8 2336.45  4776.0 2332.56  4781.9 2332.92  4818.2 2327.36  4862.9 2323.60
  4926.9 2320.11  4942.1 2318.63  4948.0 2316.96  4993.5 2314.59  4998.5 2312.82
  4999.0 2312.32  5005.1 2312.82  5034.7 2315.36  5042.6 2317.95  5084.3 2339.66
  5113.0 2348.62  5127.4 2351.92  5136.8 2352.85  5170.5 2357.26  5272.0 2360.28
#Mann=5,-1,0
  4534.8    0.07       0  4564.0    0.16       0  4998.5    0.07       0
  5005.1    0.16       0  5136.8    0.07       0
Bank Sta=4998.5,5005.1
Exp/Cntr=0.3,0.1

Type RM Length L Ch R = 1,25423,115,115,115
BEGIN DESCRIPTION:
Little Elm Creek 2 25423.2
END DESCRIPTION:
XS GIS Cut Line= 3
      1498727.37      6763395.46      1499091.96      6763129.83
      1499221.09      6762995.53
#Sta/Elev= 30
  4547.8 2356.95  4580.9 2355.17  4608.2 2352.46  4622.6 2351.03  4666.6 2340.56
  4693.7 2336.82  4716.8 2331.68  4730.5 2330.34  4737.7 2328.37  4767.1 2325.11
  4802.6 2322.69  4965.6 2314.04  4980.3 2310.44  4985.5 2306.12  4986.0 2305.62
  4992.1 2306.12  5003.6 2306.48  5016.4 2314.01  5023.6 2317.06  5030.5 2322.90
  5037.7 2325.73  5044.7 2332.89  5051.9 2335.06  5058.8 2342.06  5066.0 2343.43
  5073.0 2346.74  5087.1 2350.51  5115.4 2355.19  5164.1 2356.90  5185.2 2358.50
#Mann=5,-1,0
  4547.8    0.07       0  4608.2    0.16       0  4985.5    0.07       0
  4992.1    0.16       0  5164.1    0.07       0
Bank Sta=4985.5,4992.1
Exp/Cntr=0.3,0.1

Type RM Length L Ch R = 1,25308,229,229,229
BEGIN DESCRIPTION:
Little Elm Creek 2 25307.699
END DESCRIPTION:
XS GIS Cut Line= 3
      1498855.01      6763537.99      1499144.21      6763228.33
      1499287.25      6763064.75
#Sta/Elev= 30
  4576.3 2357.28  4601.7 2355.34  4625.9 2351.78  4640.0 2348.44  4661.0 2341.40
  4703.5 2330.53  4725.0 2326.96  4746.0 2324.62  4866.2 2315.78  4873.5 2315.94
  4894.6 2313.61  4951.2 2312.34  4976.3 2307.69  4976.8 2307.19  4982.9 2307.69
  4993.7 2309.96  4996.9 2313.75  5003.5 2313.75  5007.9 2315.20  5014.6 2320.43
  5022.2 2322.12  5028.8 2327.84  5036.4 2330.44  5043.1 2336.66  5050.7 2337.52
  5057.3 2340.27  5100.0 2351.04  5128.5 2355.14  5171.3 2358.55  5217.3 2358.94
#Mann=5,-1,0
  4576.3    0.07       0  4601.7    0.16       0  4976.3    0.07       0
  4982.9    0.16       0  5171.3    0.07       0
Bank Sta=4976.3,4982.9
Exp/Cntr=0.3,0.1

Type RM Length L Ch R = 1,25079,98,98,98
BEGIN DESCRIPTION:
Little Elm Creek 2 25078.98
END DESCRIPTION:
XS GIS Cut Line= 3
      1498901.90      6763614.18      1499167.48      6763452.75
      1499362.55      6763192.66
#Sta/Elev= 30
  4687.1 2358.35  4700.8 2358.12  4714.3 2357.08  4723.9 2357.45  4737.5 2354.41
  4745.3 2354.03  4760.7 2351.51  4782.1 2344.78  4809.2 2333.71  4831.2 2328.09
  4861.5 2322.92  4877.0 2321.18  4971.6 2313.12  4977.8 2308.56  4994.4 2306.95
  4994.9 2306.45  5001.0 2306.95  5006.1 2308.65  5041.5 2311.64  5070.7 2311.79
  5091.5 2310.03  5106.1 2310.47  5164.4 2324.68  5170.7 2328.03  5178.8 2330.32
  5191.5 2336.14  5220.7 2342.40  5249.8 2350.40  5285.3 2354.90  5323.0 2357.68
#Mann=4,-1,0
  4687.1    0.07       0  4700.8    0.16       0  4994.4    0.07       0
  5001.0    0.16       0
Bank Sta=4994.4,5001
Exp/Cntr=0.3,0.1

Type RM Length L Ch R = 1,24981,173,173,173
BEGIN DESCRIPTION:
Little Elm Creek 2 24980.58
END DESCRIPTION:
XS GIS Cut Line= 3
      1499029.48      6763762.62      1499243.01      6763515.25
      1499414.88      6763254.83
#Sta/Elev= 30
  4680.2 2358.99  4748.6 2355.95  4758.2 2355.27  4779.1 2350.31  4786.7 2346.66
  4793.4 2345.77  4815.3 2336.83  4858.0 2324.33  4885.5 2319.16  4929.4 2314.88
  4956.8 2312.69  4963.7 2310.83  4971.0 2307.11  4988.6 2304.73  4989.1 2304.23
  4995.3 2304.73  5027.6 2309.78  5051.5 2308.86  5071.9 2308.36  5092.9 2309.70
  5129.0 2314.35  5135.5 2316.21  5150.1 2317.22  5165.2 2319.93  5186.2 2326.41
  5216.4 2339.09  5231.3 2341.99  5243.4 2345.96  5273.6 2352.22  5319.0 2355.97
#Mann=6,-1,0
  4680.2    0.07       0  4748.6    0.16       0  4929.4    0.07       0
  4988.6    0.07       0  4995.3    0.07       0  5051.5    0.16       0
Bank Sta=4988.6,4995.3
Exp/Cntr=0.3,0.1

Type RM Length L Ch R = 1,24808,282,282,282
BEGIN DESCRIPTION:
Little Elm Creek 2 24808.168
END DESCRIPTION:
XS GIS Cut Line= 3
      1499255.01      6763837.98      1499378.51      6763611.00
      1499455.00      6763338.01
#Sta/Elev= 30
  4741.6 2355.66  4755.3 2354.68  4764.3 2352.07  4793.3 2340.24  4816.0 2332.81
  4821.3 2329.93  4831.3 2327.45  4844.0 2322.93  4866.8 2317.93  4924.4 2312.55
  4956.7 2311.04  4978.6 2305.29  4995.5 2304.11  4996.0 2303.61  5002.2 2304.11
  5023.9 2308.09  5080.3 2310.11  5086.2 2311.10  5133.8 2314.29  5148.5 2315.09
  5169.3 2317.41  5179.7 2318.63  5187.8 2320.46  5193.0 2321.73  5210.8 2328.43
  5227.2 2335.76  5261.3 2344.09  5266.5 2344.71  5280.9 2349.54  5283.5 2349.54
#Mann=5,-1,0
  4741.6    0.16       0  4816.0    0.07       0  4995.5    0.07       0
  5002.2    0.07       0  5133.8    0.16       0
Bank Sta=4995.5,5002.2
Exp/Cntr=0.3,0.1

Type RM Length L Ch R = 1,24526,130,130,130
BEGIN DESCRIPTION:
Little Elm Creek 2 24526.04
END DESCRIPTION:
XS GIS Cut Line= 3
      1499292.51      6763968.35      1499584.15      6763762.64
      1499826.33      6763476.19
#Sta/Elev= 30
  4646.1 2357.63  4674.2 2356.89  4711.9 2355.67  4734.8 2352.50  4786.4 2335.57
  4827.7 2321.55  4848.6 2315.89  4863.4 2313.55  4920.1 2309.04  4949.6 2303.15
  4970.6 2303.57  4981.9 2302.56  4982.4 2302.06  4988.7 2302.56  5000.1 2305.69
  5028.1 2304.39  5063.3 2309.68  5105.3 2313.52  5169.8 2318.70  5219.3 2324.48
  5255.6 2330.76  5290.7 2338.87  5311.6 2340.82  5325.9 2343.34  5333.6 2345.55
  5340.2 2345.81  5347.9 2348.12  5368.7 2351.12  5373.6 2352.50  5378.1 2352.50
#Mann=6,-1,0
  4646.1    0.07       0  4674.2    0.16       0  4786.4    0.07       0
  4981.9    0.07       0  4988.7    0.07       0  5105.3    0.16       0
Bank Sta=4981.9,4988.7
Exp/Cntr=0.3,0.1

Type RM Length L Ch R = 1,24396,134,134,134
BEGIN DESCRIPTION:
Little Elm Creek 2 24396.26
END DESCRIPTION:
XS GIS Cut Line= 3
      1499326.31      6764069.95      1499638.84      6763877.23
      1500015.43      6763612.32
#Sta/Elev= 30
  4631.3 2356.54  4667.3 2356.28  4703.9 2354.50  4725.2 2350.92  4734.7 2347.24
  4740.6 2346.92  4756.0 2341.76  4761.9 2341.46  4808.8 2328.11  4835.2 2323.13
  4841.2 2321.03  4877.8 2314.70  4929.8 2309.06  4951.1 2308.06  4958.7 2306.95
  4972.4 2301.60  4999.5 2300.45  5000.0 2299.95  5006.3 2300.45  5011.5 2301.77
  5030.5 2304.06  5067.1 2302.34  5110.0 2311.30  5175.3 2315.30  5238.3 2326.26
  5267.7 2328.91  5311.7 2335.23  5404.5 2352.15  5439.8 2355.53  5458.9 2357.39
#Mann=7,-1,0
  4631.3    0.07       0  4667.3    0.16       0  4808.8    0.07       0
  4999.5    0.07       0  5006.3    0.07       0  5011.5    0.16       0
  5439.8    0.07       0
Bank Sta=4999.5,5006.3
Exp/Cntr=0.3,0.1

Type RM Length L Ch R = 1,24262,107,107,107
BEGIN DESCRIPTION:
Little Elm Creek 2 24261.78
END DESCRIPTION:
XS GIS Cut Line= 3
      1499375.85      6764127.21      1499703.94      6763989.20
      1500060.39      6763749.84
#Sta/Elev= 30
  4641.7 2353.45  4673.1 2349.75  4678.5 2350.34  4684.2 2347.42  4702.3 2344.03
  4731.5 2341.88  4749.3 2338.65  4755.2 2335.48  4760.6 2335.47  4778.9 2330.58
  4797.9 2327.30  4825.2 2320.89  4868.6 2315.11  4964.4 2307.16  4990.6 2304.64
  4995.5 2302.71  5018.4 2298.43  5018.9 2297.93  5025.2 2298.43  5035.0 2301.08
  5048.9 2302.64  5093.8 2301.16  5135.9 2311.53  5143.5 2310.76  5192.9 2315.71
  5243.9 2323.39  5288.0 2328.36  5294.9 2330.68  5315.9 2333.06  5427.0 2354.95
#Mann=5,-1,0
  4641.7    0.16       0  4797.9    0.07       0  4964.4    0.16       0
  5018.4    0.07       0  5025.2    0.16       0
Bank Sta=5018.4,5025.2
Exp/Cntr=0.3,0.1

Type RM Length L Ch R = 1,24155,255,255,255
BEGIN DESCRIPTION:
Little Elm Creek 2 24154.88
END DESCRIPTION:
XS GIS Cut Line= 3
      1499420.09      6764194.93      1499792.48      6764059.52
      1500146.64      6763900.67
#Sta/Elev= 30
  4615.5 2342.14  4654.2 2340.02  4673.9 2336.65  4679.5 2334.42  4684.8 2335.45
  4704.7 2332.83  4710.1 2333.26  4735.3 2327.45  4740.6 2327.84  4761.0 2325.09
  4801.8 2320.61  4844.2 2314.00  4913.6 2307.38  4955.4 2304.83  4974.7 2303.84
  5000.0 2299.13  5020.4 2298.45  5020.9 2297.95  5027.2 2298.45  5029.3 2300.24
  5047.0 2301.20  5113.1 2300.53  5135.1 2308.72  5173.9 2317.10  5248.9 2328.05
  5266.6 2332.33  5277.5 2337.13  5323.9 2344.94  5376.3 2356.32  5399.9 2357.41
#Mann=6,-1,0
  4615.5    0.16       0  4761.0    0.07       0  4955.4    0.16       0
  5020.4    0.07       0  5027.2    0.16       0  5376.3    0.07       0
Bank Sta=5020.4,5027.2
Exp/Cntr=0.3,0.1

Type RM Length L Ch R = 1,23900,134,134,134
BEGIN DESCRIPTION:
Little Elm Creek 2 23900.33
END DESCRIPTION:
XS GIS Cut Line= 3
      1499443.50      6764234.00      1499948.73      6764249.62
      1500185.67      6764213.17
#Sta/Elev= 30
  4489.8 2333.29  4521.7 2329.80  4614.0 2319.39  4651.4 2317.26  4671.4 2314.51
  4721.4 2312.12  4748.7 2308.81  4778.4 2306.99  4881.5 2300.63  4941.5 2299.03
  4961.5 2297.48  4978.1 2293.62  4978.6 2293.12  4984.9 2293.62  4995.3 2293.74
  5001.6 2299.75  5011.7 2306.43  5021.8 2310.62  5032.0 2312.41  5037.9 2314.98
  5043.0 2315.21  5062.3 2320.58  5072.4 2322.13  5082.6 2325.61  5106.2 2329.20
  5169.5 2341.65  5174.5 2341.58  5204.0 2349.50  5222.4 2352.98  5235.0 2354.67
#Mann=8,-1,0
  4489.8    0.16       0  4521.7    0.07       0  4614.0    0.16       0
  4748.7    0.07       0  4778.4    0.16       0  4978.1    0.07       0
  4984.9    0.16       0  5222.4    0.07       0
Bank Sta=4978.1,4984.9
Exp/Cntr=0.3,0.1

Type RM Length L Ch R = 1,23766,356,356,356
BEGIN DESCRIPTION:
Little Elm Creek 2 23766.12
END DESCRIPTION:
XS GIS Cut Line= 3
      1499430.46      6764325.14      1499917.48      6764369.41
      1500117.97      6764468.35
#Sta/Elev= 30
  4506.1 2340.77  4530.7 2338.29  4560.9 2331.79  4593.7 2326.69  4601.0 2324.41
  4641.0 2320.01  4761.7 2306.08  4810.4 2302.91  4832.0 2299.04  4902.3 2298.80
  4962.5 2296.75  4995.1 2293.81  4997.2 2292.10  4997.7 2291.60  5004.0 2292.10
  5006.2 2292.53  5023.0 2303.75  5037.0 2309.83  5073.5 2314.65  5090.4 2318.41
  5096.0 2318.33  5126.2 2325.64  5148.5 2328.72  5157.7 2331.27  5163.3 2331.20
  5180.2 2335.03  5185.8 2334.78  5193.1 2337.25  5209.1 2339.70  5218.7 2341.51
#Mann=6,-1,0
  4506.1    0.16       0  4593.7    0.07       0  4641.0    0.16       0
  4997.2    0.07       0  5004.0    0.16       0  5209.1    0.07       0
Bank Sta=4997.2,5004
Exp/Cntr=0.3,0.1

Type RM Length L Ch R = 1,23410,159,159,159
BEGIN DESCRIPTION:
Little Elm Creek 2 23409.87
END DESCRIPTION:
XS GIS Cut Line= 3
      1499328.99      6764541.28      1499651.86      6764510.04
      1500084.13      6764564.72
#Sta/Elev= 30
  4673.2 2344.91  4702.0 2341.62  4739.5 2337.89  4749.6 2334.90  4756.9 2330.15
  4761.9 2330.77  4779.7 2322.13  4789.8 2320.09  4859.0 2316.26  4864.1 2317.21
  4950.5 2310.82  4960.5 2306.92  4966.2 2298.48  4971.2 2302.92  4980.6 2291.74
  5018.5 2291.15  5020.1 2288.74  5020.6 2288.24  5027.0 2288.74  5041.1 2293.84
  5098.7 2300.53  5173.7 2301.74  5212.4 2304.00  5259.0 2310.21  5333.4 2312.11
  5339.2 2314.47  5344.2 2314.32  5363.6 2321.23  5419.3 2334.91  5433.3 2336.63
#Mann=5,-1,0
  4673.2    0.16       0  4702.0    0.07       0  5020.1    0.07       0
  5027.0    0.07       0  5173.7    0.16       0
Bank Sta=5020.1,5027
Exp/Cntr=0.3,0.1

Type RM Length L Ch R = 1,23251,107,107,107
BEGIN DESCRIPTION:
Little Elm Creek 2 23251.32
END DESCRIPTION:
XS GIS Cut Line= 3
      1499315.88      6764668.89      1499659.67      6764668.89
      1500058.07      6764629.83
#Sta/Elev= 30
  4662.1 2337.49  4682.1 2335.70  4721.2 2332.34  4771.2 2326.68  4861.2 2319.56
  4901.2 2313.24  4931.2 2310.70  4941.2 2309.15  4951.2 2301.67  4971.2 2288.42
  4987.8 2286.62  4988.3 2286.12  4994.7 2286.62  5005.9 2286.64  5011.2 2289.11
  5021.3 2290.13  5041.4 2298.38  5051.4 2299.66  5122.5 2302.79  5172.9 2304.95
  5192.1 2308.51  5212.2 2310.05  5282.5 2310.21  5322.7 2311.31  5332.8 2312.89
  5370.8 2323.58  5375.9 2322.87  5383.0 2325.87  5402.2 2329.01  5406.2 2329.01
#Mann=5,-1,0
  4662.1    0.16       0  4682.1    0.07       0  4987.8    0.07       0
  4994.7    0.07       0  5122.5    0.16       0
Bank Sta=4987.8,4994.7
Exp/Cntr=0.3,0.1

Type RM Length L Ch R = 1,23144,171,171,171
BEGIN DESCRIPTION:
Little Elm Creek 2 23144.24
END DESCRIPTION:
XS GIS Cut Line= 3
      1499313.31      6764754.83      1499597.17      6764760.04
      1499904.42      6764765.25
#Sta/Elev= 30
  4708.0 2329.06  4780.5 2325.33  4789.7 2325.29  4809.7 2322.09  4829.7 2320.55
  4839.7 2319.17  4859.7 2318.44  4879.7 2315.91  4919.7 2312.32  4949.7 2311.23
  4979.7 2308.69  4988.3 2300.03  4991.9 2300.03  4999.7 2290.61  5009.7 2285.77
  5016.3 2284.79  5016.8 2284.29  5022.7 2284.29  5023.2 2284.79  5039.7 2288.94
  5049.7 2289.24  5059.7 2290.70  5069.8 2294.74  5089.8 2298.48  5146.0 2301.30
  5170.7 2303.06  5209.8 2304.60  5249.8 2307.37  5279.8 2307.42  5299.2 2308.60
#Mann=5,-1,0
  4708.0    0.16       0  4780.5    0.07       0  5016.3    0.07       0
  5023.2    0.07       0  5146.0    0.16       0
Bank Sta=5016.3,5023.2
Exp/Cntr=0.3,0.1

Type RM Length L Ch R = 1,22973,120,120,120
BEGIN DESCRIPTION:
Little Elm Creek 2 22973.47
END DESCRIPTION:
XS GIS Cut Line= 3
      1499162.26      6764869.41      1499610.19      6764885.04
      1499956.59      6764861.60
#Sta/Elev= 30
  4549.7 2322.47  4582.5 2322.32  4622.5 2320.95  4642.5 2319.94  4662.5 2317.51
  4722.5 2316.02  4762.6 2316.18  4780.2 2315.54  4832.6 2313.61  4862.6 2311.52
  4938.6 2308.10  4952.7 2305.36  4972.7 2294.92  4982.7 2290.64  4994.4 2289.56
  4994.9 2289.06  5000.8 2289.06  5001.3 2289.56  5022.8 2289.60  5041.2 2291.55
  5062.9 2295.60  5115.4 2297.69  5133.0 2300.96  5143.0 2301.70  5193.2 2304.58
  5283.4 2308.05  5324.5 2312.89  5333.5 2313.47  5341.8 2315.33  5345.1 2315.33
#Mann=7,-1,0
  4549.7    0.16       0  4780.2    0.07       0  4994.4    0.07       0
  5001.3    0.07       0  5041.2    0.16       0  5115.4    0.07       0
  5324.5    0.16       0
Bank Sta=4994.4,5001.3
Exp/Cntr=0.3,0.1

Type RM Length L Ch R = 1,22853,268,268,268
BEGIN DESCRIPTION:
Little Elm Creek 2 22852.54
END DESCRIPTION:
XS GIS Cut Line= 3
      1499164.87      6764960.56      1499607.59      6765004.83
      1499940.46      6764986.63
#Sta/Elev= 30
  4558.3 2311.68  4608.7 2308.74  4678.7 2308.74  4683.7 2308.03  4784.2 2309.03
  4839.8 2307.27  4870.0 2304.56  4884.7 2304.12  4890.1 2303.12  4930.3 2299.99
  4940.3 2297.95  4960.4 2291.22  4980.2 2286.39  4985.2 2286.82  4987.1 2285.70
  4987.6 2285.20  4993.5 2285.20  4994.0 2285.70  5010.7 2287.08  5036.2 2292.01
  5070.7 2295.16  5120.8 2298.40  5140.8 2300.24  5190.9 2302.83  5217.9 2305.09
  5241.0 2305.17  5271.0 2307.48  5281.1 2307.62  5311.1 2310.58  5336.6 2314.60
#Mann=3,-1,0
  4558.3    0.07       0  4987.1    0.07       0  4994.0    0.07       0
Bank Sta=4987.1,4994
Exp/Cntr=0.3,0.1

Type RM Length L Ch R = 1,22585,127,127,127
BEGIN DESCRIPTION:
Little Elm Creek 2 22584.52
END DESCRIPTION:
XS GIS Cut Line= 3
      1499177.94      6765228.79      1499604.98      6765226.18
      1500016.40      6765158.48
#Sta/Elev= 30
  4570.0 2318.21  4597.1 2315.15  4787.1 2308.02  4827.1 2305.20  4857.1 2304.58
  4877.1 2301.86  4897.5 2300.49  4898.0 2300.45  4937.1 2296.26  4947.1 2294.10
  4957.1 2284.32  4963.5 2282.65  4964.0 2282.15  4970.7 2282.65  5019.5 2286.21
  5037.6 2291.19  5047.7 2292.24  5057.9 2291.91  5068.0 2288.61  5088.3 2289.68
  5098.4 2293.13  5108.5 2295.18  5165.9 2300.17  5198.7 2303.58  5264.3 2306.90
  5320.4 2313.98  5372.0 2316.37  5381.6 2317.59  5386.7 2317.12  5414.0 2320.99
#Mann=7,-1,0
  4570.0    0.07       0  4897.5    0.16       0  4898.0    0.07       0
  4963.5    0.07       0  4970.7    0.07       0  5165.9    0.16       0
  5198.7    0.07       0
Bank Sta=4963.5,4970.7
Exp/Cntr=0.3,0.1

Type RM Length L Ch R = 1,22458,195,195,195
BEGIN DESCRIPTION:
Little Elm Creek 2 22457.61
END DESCRIPTION:
XS GIS Cut Line= 3
      1499355.00      6765330.35      1499651.86      6765338.16
      1499969.60      6765299.10
#Sta/Elev= 30
  4700.7 2310.66  4730.7 2308.45  4750.7 2308.76  4770.7 2307.05  4790.7 2307.21
  4803.6 2304.84  4841.0 2300.61  4879.1 2296.16  4910.8 2294.06  4920.8 2292.51
  4930.8 2281.87  4940.8 2277.70  4947.2 2276.88  4947.7 2276.38  4953.9 2276.38
  4954.4 2276.88  4960.8 2277.58  4970.8 2279.91  4990.8 2280.40  4996.7 2283.86
  5001.8 2283.86  5031.1 2289.56  5071.4 2291.77  5097.7 2295.46  5119.3 2299.04
  5190.8 2306.18  5242.6 2310.22  5286.9 2312.18  5293.0 2313.24  5317.8 2313.94
#Mann=7,-1,0
  4700.7    0.07       0  4841.0    0.16       0  4879.1    0.07       0
  4947.2    0.07       0  4954.4    0.07       0  5097.7    0.16       0
  5190.8    0.07       0
Bank Sta=4947.2,4954.4
Exp/Cntr=0.3,0.1

Type RM Length L Ch R = 1,22263,108,108,108
BEGIN DESCRIPTION:
Little Elm Creek 2 22263.07
END DESCRIPTION:
XS GIS Cut Line= 3
      1499347.18      6765455.35      1499753.42      6765489.20
      1500026.83      6765439.73
#Sta/Elev= 30
  4598.6 2309.10  4656.6 2305.97  4676.7 2303.47  4686.2 2300.84  4691.2 2300.87
  4696.8 2299.30  4727.7 2297.58  4787.1 2297.62  4827.2 2296.15  4857.3 2292.38
  4867.4 2291.83  4887.4 2288.69  4927.0 2279.30  4957.7 2277.98  4983.0 2275.71
  4984.1 2275.65  4984.6 2275.15  4991.4 2275.65  5004.5 2290.55  5009.6 2290.55
  5018.0 2297.78  5028.2 2299.81  5042.3 2300.75  5058.7 2303.14  5119.6 2307.23
  5170.5 2309.38  5200.9 2311.70  5207.8 2312.83  5221.3 2312.74  5284.1 2315.74
#Mann=5,-1,0
  4598.6    0.07       0  4727.7    0.16       0  4983.0    0.07       0
  4984.1    0.07       0  4991.4    0.07       0
Bank Sta=4984.1,4991.4
Exp/Cntr=0.3,0.1

Type RM Length L Ch R = 1,22155,145,145,145
BEGIN DESCRIPTION:
Little Elm Creek 2 22155.24
END DESCRIPTION:
XS GIS Cut Line= 3
      1499326.37      6765556.91      1499703.94      6765582.95
      1500031.01      6765569.98
#Sta/Elev= 30
  4620.9 2308.39  4639.6 2308.17  4699.7 2305.26  4707.0 2303.77  4712.1 2303.83
  4721.1 2302.63  4749.8 2298.69  4769.9 2297.38  4849.9 2296.67  4907.9 2291.42
  4950.3 2287.59  4997.4 2278.24  5002.4 2278.24  5013.1 2274.26  5016.8 2273.24
  5017.3 2272.74  5023.6 2272.74  5024.1 2273.24  5030.5 2275.19  5060.5 2287.16
  5070.5 2293.34  5080.5 2297.74  5083.4 2298.41  5110.5 2303.50  5160.6 2307.28
  5200.6 2308.31  5253.0 2311.91  5280.7 2312.52  5300.7 2313.70  5326.7 2313.64
#Mann=7,-1,0
  4620.9    0.07       0  4721.1    0.16       0  4907.9    0.07       0
  5013.1    0.16       0  5016.8    0.07       0  5024.1    0.16       0
  5083.4    0.07       0
Bank Sta=5016.8,5024.1
Exp/Cntr=0.3,0.1

Type RM Length L Ch R = 1,22010,207,207,207
BEGIN DESCRIPTION:
Little Elm Creek 2 22009.79
END DESCRIPTION:
XS GIS Cut Line= 3
      1499321.17      6765666.29      1499750.82      6765713.16
      1500045.11      6765666.28
#Sta/Elev= 30
  4563.9 2306.85  4614.6 2304.56  4648.2 2303.99  4678.4 2300.41  4715.8 2299.37
  4738.8 2296.81  4779.0 2293.73  4859.5 2289.95  4869.5 2288.74  4898.5 2281.38
  4950.0 2279.56  4976.5 2272.35  4977.0 2271.85  4983.8 2272.35  4989.9 2273.53
  4994.9 2278.59  5001.3 2279.48  5010.5 2293.43  5020.6 2296.87  5038.7 2298.68
  5058.4 2300.39  5063.4 2300.14  5071.2 2302.05  5101.6 2305.63  5132.0 2307.40
  5170.0 2308.15  5187.7 2309.39  5233.2 2310.05  5243.4 2311.57  5294.1 2312.52
#Mann=6,-1,0
  4563.9    0.07       0  4614.6    0.16       0  4976.5    0.07       0
  4983.8    0.16       0  5038.7    0.07       0  5170.0   0.035       0
Bank Sta=4976.5,4983.8
Exp/Cntr=0.3,0.1

Type RM Length L Ch R = 1,21803,260,260,260
BEGIN DESCRIPTION:
Little Elm Creek 2 21802.75
END DESCRIPTION:
XS GIS Cut Line= 3
      1499263.84      6765942.33      1499711.76      6765903.27
      1500001.72      6765825.60
#Sta/Elev= 30
  4557.3 2311.39  4689.0 2303.60  4709.0 2300.97  4789.3 2296.39  4819.5 2292.16
  4849.6 2289.36  4869.6 2286.20  4889.7 2285.01  4894.8 2283.23  4899.8 2283.65
  4939.9 2276.39  4970.0 2275.95  5002.3 2271.05  5002.8 2270.55  5009.7 2271.05
  5014.0 2271.69  5020.6 2272.14  5031.0 2274.99  5041.3 2275.53  5046.6 2278.71
  5051.7 2278.11  5072.4 2286.70  5093.1 2292.23  5117.2 2295.10  5175.9 2300.31
  5196.3 2300.66  5220.4 2304.03  5227.7 2304.31  5236.3 2302.98  5307.1 2306.05
#Mann=6,-1,0
  4557.3    0.07       0  5002.3    0.07       0  5009.7    0.07       0
  5014.0    0.16       0  5117.2    0.07       0  5220.4   0.035       0
Bank Sta=5002.3,5009.7
Exp/Cntr=0.3,0.1

Type RM Length L Ch R = 1,21543,181,181,181
BEGIN DESCRIPTION:
Little Elm Creek 2 21543.28
END DESCRIPTION:
XS GIS Cut Line= 3
      1499321.17      6766137.64      1499662.28      6766148.06
      1499949.32      6765982.56
#Sta/Elev= 30
  4666.7 2309.60  4707.5 2306.96  4720.6 2306.48  4740.6 2302.87  4760.6 2300.83
  4800.6 2301.20  4870.6 2299.71  4940.7 2291.50  4960.7 2290.95  4970.7 2289.05
  4990.7 2278.52  5000.7 2271.89  5003.1 2267.69  5003.6 2267.19  5010.5 2267.69
  5017.5 2270.23  5033.3 2271.96  5054.8 2272.49  5068.8 2270.62  5076.4 2273.81
  5097.9 2276.87  5113.7 2276.66  5149.6 2278.78  5194.2 2283.51  5199.9 2282.44
  5221.5 2283.64  5280.4 2291.47  5323.5 2293.38  5333.5 2292.60  5339.3 2293.60
#Mann=4,-1,0
  4666.7    0.07       0  4707.5   0.035       0  5003.1   0.035       0
  5010.5   0.035       0
Bank Sta=5003.1,5010.5
Exp/Cntr=0.3,0.1

Type RM Length L Ch R = 1,21362,143,143,143
BEGIN DESCRIPTION:
Little Elm Creek 2 21361.55
END DESCRIPTION:
XS GIS Cut Line= 3
      1499568.51      6766452.76      1499782.07      6766257.43
      1499960.90      6765998.26
#Sta/Elev= 30
  4717.0 2312.61  4767.2 2308.22  4788.8 2307.18  4809.7 2303.70  4823.9 2301.92
  4838.1 2301.04  4923.2 2289.72  4930.0 2288.26  4944.2 2275.57  4951.6 2271.83
  4958.3 2270.53  4979.9 2268.83  4990.4 2265.84  4990.9 2265.34  4997.3 2265.34
  4997.8 2265.84  5000.9 2269.26  5005.0 2272.71  5009.1 2272.71  5016.1 2274.35
  5033.1 2274.66  5053.0 2275.61  5087.8 2278.30  5149.9 2281.53  5188.0 2284.75
  5216.2 2285.83  5224.4 2287.17  5252.0 2289.60  5296.7 2291.21  5321.3 2293.16
#Mann=6,-1,0
  4717.0    0.07       0  4990.4    0.07       0  4997.8    0.07       0
  5033.1    0.16       0  5053.0    0.07       0  5149.9   0.035       0
Bank Sta=4990.4,4997.8
Exp/Cntr=0.3,0.1

Type RM Length L Ch R = 1,21219,181,181,181
BEGIN DESCRIPTION:
Little Elm Creek 2 21219.46
END DESCRIPTION:
XS GIS Cut Line= 3
      1499701.31      6766510.06      1499847.17      6766379.83
      1499948.73      6766049.11
#Sta/Elev= 30
  4803.8 2308.28  4822.2 2307.51  4843.3 2305.80  4857.6 2304.18  4864.3 2302.38
  4871.8 2301.85  4900.2 2297.64  4956.2 2292.59  4963.7 2288.96  4970.4 2282.83
  4977.9 2278.66  4984.6 2273.29  4997.0 2270.35  5002.9 2270.35  5007.7 2268.05
  5013.0 2266.85  5018.4 2266.50  5018.9 2266.00  5025.4 2266.00  5025.9 2266.50
  5046.1 2269.01  5064.0 2270.84  5111.1 2280.50  5147.7 2280.27  5209.3 2280.70
  5249.3 2283.95  5312.7 2287.64  5317.9 2287.42  5336.0 2290.04  5345.3 2290.55
#Mann=6,-1,0
  4803.8    0.07       0  5018.4    0.07       0  5025.9    0.07       0
  5046.1    0.16       0  5147.7    0.07       0  5249.3   0.035       0
Bank Sta=5018.4,5025.9
Exp/Cntr=0.3,0.1

Type RM Length L Ch R = 1,21038,169,169,169
BEGIN DESCRIPTION:
Little Elm Creek 2 21038.1
END DESCRIPTION:
XS GIS Cut Line= 3
      1500024.25      6766580.37      1500026.86      6766387.64
      1499966.96      6766043.87
#Sta/Elev= 30
  4807.7 2293.20  4840.1 2293.30  4900.1 2292.08  4930.1 2290.68  4940.1 2289.01
  4950.1 2284.71  4970.1 2270.41  4980.1 2265.05  4986.3 2262.87  4986.8 2262.37
  4993.3 2262.37  4993.8 2262.87  4997.8 2265.35  5020.4 2266.13  5030.5 2267.70
  5043.1 2268.86  5050.8 2272.63  5061.0 2275.44  5071.1 2277.31  5126.5 2278.12
  5152.1 2278.13  5203.1 2279.20  5223.4 2281.40  5249.2 2282.49  5264.0 2283.18
  5276.3 2284.59  5294.5 2285.25  5324.9 2288.37  5330.8 2289.82  5349.4 2290.89
#Mann=5,-1,0
  4807.7    0.16       0  4986.3    0.07       0  4993.8    0.16       0
  5126.5    0.07       0  5249.2   0.035       0
Bank Sta=4986.3,4993.8
Exp/Cntr=0.3,0.1

Type RM Length L Ch R = 1,20869,123,123,123
BEGIN DESCRIPTION:
Little Elm Creek 2 20869.36
END DESCRIPTION:
XS GIS Cut Line= 3
      1500248.20      6766442.31      1500128.42      6766275.66
      1499992.99      6766038.65
#Sta/Elev= 30
  4787.1 2282.38  4799.9 2281.83  4806.0 2282.64  4835.5 2283.40  4869.7 2283.39
  4885.8 2282.88  4900.5 2281.11  4906.7 2276.21  4915.2 2275.35  4921.4 2271.04
  4927.9 2270.21  4936.1 2267.67  4942.3 2263.53  4950.8 2264.12  4957.0 2263.00
  4986.5 2263.86  4991.0 2262.82  5001.2 2262.85  5004.4 2261.96  5004.9 2261.46
  5011.9 2261.96  5023.9 2264.51  5029.7 2271.93  5051.3 2274.38  5058.7 2273.86
  5147.8 2278.66  5212.5 2284.58  5229.6 2287.12  5250.0 2289.90  5265.3 2290.77
#Mann=5,-1,0
  4787.1    0.07       0  4869.7    0.16       0  5004.4    0.07       0
  5011.9    0.16       0  5229.6   0.035       0
Bank Sta=5004.4,5011.9
Exp/Cntr=0.3,0.1

Type RM Length L Ch R = 1,20746,206,206,206
BEGIN DESCRIPTION:
Little Elm Creek 2 20746.17
END DESCRIPTION:
XS GIS Cut Line= 3
      1500282.06      6766314.71      1500183.11      6766168.89
      1500069.28      6765959.34
#Sta/Elev= 30
  4816.6 2281.03  4876.4 2280.68  4891.3 2277.85  4897.4 2278.30  4906.3 2274.99
  4912.3 2271.13  4927.3 2265.60  4948.3 2265.95  4978.2 2264.26  4984.2 2261.39
  4996.1 2261.19  5005.2 2259.33  5011.8 2259.03  5012.3 2258.53  5019.3 2259.03
  5037.5 2266.17  5043.1 2271.26  5050.7 2272.96  5065.0 2274.50  5081.2 2274.55
  5096.3 2276.04  5119.0 2281.68  5124.9 2284.78  5141.0 2289.71  5146.7 2290.60
  5153.2 2293.22  5162.9 2295.11  5172.6 2295.22  5198.7 2296.05  5231.3 2298.40
#Mann=4,-1,0
  4816.6    0.16       0  5011.8    0.07       0  5019.3    0.16       0
  5172.6    0.07       0
Bank Sta=5011.8,5019.3
Exp/Cntr=0.3,0.1

Type RM Length L Ch R = 1,20540,232,232,232
BEGIN DESCRIPTION:
Little Elm Creek 2 20540.38
END DESCRIPTION:
XS GIS Cut Line= 3
      1500305.50      6766322.54      1500313.32      6766043.89
      1500276.86      6765793.90
#Sta/Elev= 30
  4714.6 2279.85  4729.1 2279.97  4749.2 2278.68  4779.2 2273.07  4809.2 2272.03
  4839.2 2272.20  4905.7 2266.48  4919.2 2265.64  4939.2 2260.61  4949.2 2259.75
  4959.2 2257.64  4963.6 2257.77  4993.4 2257.69  4995.6 2254.95  4996.1 2254.45
  5003.1 2254.95  5015.4 2259.86  5020.5 2255.88  5029.6 2258.47  5039.7 2264.55
  5059.9 2273.87  5070.1 2279.71  5080.2 2288.42  5085.4 2296.98  5090.5 2296.58
  5100.4 2300.85  5107.7 2301.18  5140.8 2305.40  5171.1 2307.69  5246.0 2311.32
#Mann=6,-1,0
  4714.6    0.16       0  4905.7    0.07       0  4963.6    0.16       0
  4995.6    0.07       0  5003.1    0.16       0  5107.7    0.07       0
Bank Sta=4995.6,5003.1
Exp/Cntr=0.3,0.1

Type RM Length L Ch R = 1,20308,212,212,212
BEGIN DESCRIPTION:
Little Elm Creek 2 20308.3
END DESCRIPTION:
XS GIS Cut Line= 3
      1500329.99      6766313.01      1500461.76      6766194.93
      1500570.40      6765874.16
#Sta/Elev= 30
  4822.9 2279.66  4829.6 2279.35  4851.3 2273.82  4865.5 2266.58  4879.7 2262.31
  4908.1 2260.43  4914.9 2261.10  4922.4 2258.46  4929.1 2259.04  4936.6 2256.93
  4964.2 2256.99  4982.1 2254.27  4982.6 2253.77  4989.6 2254.27  5009.1 2256.78
  5017.7 2257.62  5029.5 2256.85  5070.5 2259.81  5081.1 2262.80  5087.1 2269.42
  5092.4 2278.04  5102.2 2287.34  5118.5 2289.58  5123.8 2288.81  5143.4 2291.01
  5244.2 2293.44  5270.4 2294.96  5275.6 2294.21  5301.8 2295.32  5338.5 2294.71
#Mann=5,-1,0
  4822.9    0.07       0  4982.1    0.07       0  4989.6    0.07       0
  5009.1    0.16       0  5143.4    0.07       0
Bank Sta=4982.1,4989.6
Exp/Cntr=0.3,0.1

Type RM Length L Ch R = 1,20096,235,235,235
BEGIN DESCRIPTION:
Little Elm Creek 2 20095.64
END DESCRIPTION:
XS GIS Cut Line= 3
      1500701.34      6766551.73      1500615.40      6766184.52
      1500657.07      6765853.77
#Sta/Elev= 30
  4626.8 2297.71  4654.5 2296.38  4702.5 2292.44  4761.7 2283.73  4774.4 2282.66
  4795.0 2281.28  4856.9 2279.36  4866.8 2275.59  4877.1 2268.65  4894.3 2259.37
  4907.9 2256.52  4933.9 2255.66  4977.9 2252.36  4984.2 2251.91  4984.7 2251.41
  4996.0 2251.91  5010.5 2252.19  5030.7 2261.46  5043.3 2261.30  5050.8 2262.17
  5091.1 2273.25  5111.3 2276.73  5131.5 2278.34  5198.9 2288.34  5203.9 2287.26
  5222.2 2288.89  5279.2 2291.50  5292.7 2291.46  5323.8 2293.47  5337.3 2294.07
#Mann=7,-1,0
  4626.8    0.07       0  4654.5    0.16       0  4933.9    0.07       0
  4977.9    0.16       0  4984.2    0.07       0  4996.0    0.16       0
  5323.8    0.07       0
Bank Sta=4984.2,4996
Exp/Cntr=0.3,0.1

Type RM Length L Ch R = 1,19861,163,163,163
BEGIN DESCRIPTION:
Little Elm Creek 2 19861.25
END DESCRIPTION:
XS GIS Cut Line= 3
      1500888.84      6766528.29      1500849.78      6766189.73
      1500709.59      6765805.51
#Sta/Elev= 30
  4661.7 2298.31  4775.6 2289.78  4822.0 2284.75  4827.1 2285.12  4863.3 2279.48
  4923.7 2274.97  4930.1 2268.55  4934.6 2264.35  4943.9 2258.67  4964.0 2254.15
  4974.1 2249.55  4994.0 2248.86  4994.5 2248.36  5005.8 2248.86  5031.0 2252.54
  5046.9 2253.23  5056.2 2255.63  5061.6 2255.62  5068.2 2257.92  5132.1 2257.15
  5142.6 2258.90  5164.0 2272.41  5173.1 2275.01  5234.2 2280.06  5243.7 2281.72
  5302.4 2289.61  5335.7 2291.07  5351.1 2291.50  5371.9 2293.90  5411.5 2295.85
#Mann=9,-1,0
  4661.7    0.07       0  4775.6    0.16       0  4930.1    0.07       0
  4934.6    0.16       0  4994.0    0.07       0  5005.8    0.16       0
  5243.7    0.07       0  5335.7    0.16       0  5371.9    0.07       0
Bank Sta=4994,5005.8
Exp/Cntr=0.3,0.1

Type RM Length L Ch R = 1,19698,202,202,202
BEGIN DESCRIPTION:
Little Elm Creek 2 19697.81
END DESCRIPTION:
XS GIS Cut Line= 3
      1501104.99      6766541.31      1500990.40      6766197.54
      1500834.14      6765796.48
#Sta/Elev= 30
  4628.7 2297.68  4758.7 2291.47  4793.4 2288.43  4874.6 2282.19  4937.9 2274.79
  4949.2 2270.86  4957.2 2263.60  4962.5 2262.38  4969.5 2255.15  4980.0 2250.94
  4988.1 2246.06  4988.6 2245.56  5000.0 2246.06  5012.0 2247.17  5018.6 2249.71
  5033.5 2251.10  5048.4 2252.05  5065.7 2250.61  5088.2 2256.28  5151.6 2255.66
  5162.6 2256.53  5205.2 2255.20  5211.6 2256.87  5216.9 2259.66  5236.1 2275.40
  5312.5 2278.68  5334.0 2282.00  5344.7 2282.28  5380.1 2288.51  5421.5 2290.30
#Mann=6,-1,0
  4628.7    0.07       0  4793.4    0.16       0  4949.2    0.07       0
  4988.1    0.07       0  5000.0    0.07       0  5088.2    0.16       0
Bank Sta=4988.1,5000
Exp/Cntr=0.3,0.1

Type RM Length L Ch R = 1,19496,222,222,222
BEGIN DESCRIPTION:
Little Elm Creek 2 19496.19
END DESCRIPTION:
XS GIS Cut Line= 3
      1501399.24      6766450.13      1501149.26      6766088.16
      1500966.97      6765736.61
#Sta/Elev= 30
  4567.7 2290.38  4666.7 2287.99  4702.5 2284.75  4744.4 2282.96  4759.3 2280.70
  4780.2 2280.61  4800.1 2276.32  4824.9 2273.35  4887.7 2269.19  4896.5 2263.15
  4923.6 2254.01  4938.4 2250.56  4977.1 2245.45  4977.6 2244.95  4989.0 2245.45
  4995.6 2247.16  5026.2 2247.68  5041.6 2252.33  5054.5 2253.71  5131.2 2252.15
  5159.0 2256.53  5175.4 2268.00  5181.1 2267.93  5188.0 2273.35  5197.6 2276.28
  5269.6 2276.26  5291.7 2277.75  5323.2 2280.49  5396.7 2291.33  5403.6 2291.18
#Mann=6,-1,0
  4567.7    0.07       0  4702.5    0.16       0  4800.1    0.07       0
  4977.1    0.07       0  4989.0    0.07       0  5054.5    0.16       0
Bank Sta=4977.1,4989
Exp/Cntr=0.3,0.1

Type RM Length L Ch R = 1,19274,308,308,308
BEGIN DESCRIPTION:
Little Elm Creek 2 19274.41
END DESCRIPTION:
XS GIS Cut Line= 3
      1501516.46      6766366.84      1501336.76      6765986.60
      1501043.98      6765781.92
#Sta/Elev= 30
  4582.3 2282.30  4671.3 2278.71  4711.3 2273.49  4791.2 2268.58  4830.7 2255.50
  4836.2 2256.65  4846.5 2253.40  4890.7 2250.84  4904.5 2245.26  4935.0 2247.74
  4967.2 2243.55  4972.8 2246.18  5006.0 2246.06  5018.4 2243.75  5019.0 2243.48
  5019.5 2242.98  5030.9 2243.48  5031.1 2245.36  5045.9 2252.49  5075.5 2252.33
  5090.4 2254.00  5096.5 2258.42  5111.3 2259.05  5117.4 2265.00  5126.1 2263.49
  5132.2 2270.01  5139.2 2271.52  5182.8 2275.00  5340.7 2281.10  5360.1 2283.66
#Mann=4,-1,0
  4582.3    0.07       0  5018.4    0.16       0  5019.0    0.07       0
  5030.9    0.16       0
Bank Sta=5019,5030.9
Exp/Cntr=0.3,0.1

Type RM Length L Ch R = 1,18966,209,209,209
BEGIN DESCRIPTION:
Little Elm Creek 2 18965.74
END DESCRIPTION:
XS GIS Cut Line= 3
      1501597.17      6766408.47      1501631.03      6766036.08
      1501784.01      6765621.21
#Sta/Elev= 30
  4628.1 2281.90  4661.5 2278.72  4729.0 2275.17  4789.2 2268.32  4829.4 2266.31
  4869.6 2257.95  4877.4 2254.63  4882.4 2254.68  4899.7 2249.42  4939.8 2245.75
  4949.9 2243.55  4959.9 2243.12  4981.0 2240.04  4981.5 2239.54  4994.7 2240.04
  4998.5 2241.50  5021.3 2241.87  5027.3 2246.96  5042.6 2250.08  5062.8 2249.86
  5118.6 2250.34  5127.9 2252.20  5138.4 2257.50  5143.7 2256.72  5149.2 2263.54
  5159.8 2269.91  5290.6 2276.53  5346.1 2281.04  5376.6 2285.03  5444.2 2288.99
#Mann=4,-1,0
  4628.1    0.07       0  4981.0    0.07       0  4994.7    0.07       0
  5062.8    0.16       0
Bank Sta=4981,4994.7
Exp/Cntr=0.3,0.1

Type RM Length L Ch R = 1,18757,191,191,191
BEGIN DESCRIPTION:
Little Elm Creek 2 18756.58
END DESCRIPTION:
XS GIS Cut Line= 3
      1501654.45      6766411.11      1501834.15      6766059.52
      1501960.06      6765823.12
#Sta/Elev= 30
  4610.9 2277.51  4671.6 2274.46  4777.1 2262.04  4838.1 2250.55  4850.2 2245.90
  4860.3 2244.47  4888.2 2243.17  4904.8 2245.13  4932.6 2244.35  4985.0 2239.59
  4996.9 2237.45  4997.4 2236.95  5010.7 2237.45  5015.7 2241.07  5021.3 2240.39
  5030.1 2244.74  5052.8 2244.86  5059.6 2246.29  5075.2 2246.65  5103.5 2246.33
  5119.8 2252.11  5125.5 2252.58  5132.1 2257.53  5141.8 2261.90  5163.8 2268.47
  5229.7 2273.96  5235.3 2273.21  5251.6 2276.59  5257.3 2275.91  5273.6 2277.20
#Mann=4,-1,0
  4610.9    0.07       0  4996.9    0.07       0  5010.7    0.07       0
  5075.2    0.16       0
Bank Sta=4996.9,5010.7
Exp/Cntr=0.3,0.1

Type RM Length L Ch R = 1,18566,229,229,229
BEGIN DESCRIPTION:
Little Elm Creek 2 18566.41
END DESCRIPTION:
XS GIS Cut Line= 3
      1501714.38      6766525.63      1502013.84      6766095.98
      1502060.30      6765884.33
#Sta/Elev= 30
  4479.1 2279.24  4506.5 2275.45  4521.4 2275.43  4549.3 2272.16  4658.4 2266.46
  4700.2 2261.09  4715.1 2261.00  4771.8 2251.69  4837.2 2249.52  4852.1 2247.98
  4858.2 2248.56  4866.3 2245.67  4873.0 2241.42  4887.9 2239.32  4944.6 2239.31
  4974.2 2237.61  4988.3 2235.43  4988.8 2234.93  5002.1 2235.43  5002.8 2237.42
  5011.0 2240.20  5021.2 2242.23  5034.1 2242.40  5062.2 2250.19  5077.9 2252.17
  5098.1 2253.01  5126.8 2254.10  5154.3 2260.85  5170.6 2263.42  5219.5 2266.09
#Mann=4,-1,0
  4479.1    0.07       0  4988.3    0.07       0  5002.1    0.07       0
  5098.1    0.16       0
Bank Sta=4988.3,5002.1
Exp/Cntr=0.3,0.1

Type RM Length L Ch R = 1,18337,301,301,301
BEGIN DESCRIPTION:
Little Elm Creek 2 18337.47
END DESCRIPTION:
XS GIS Cut Line= 3
      1501779.42      6766533.50      1502151.86      6766270.45
      1502396.22      6766202.87
#Sta/Elev= 30
  4540.6 2271.98  4626.4 2267.29  4657.1 2265.67  4678.1 2261.46  4713.8 2257.74
  4770.4 2254.73  4799.9 2248.05  4876.0 2247.52  4963.7 2245.13  4970.6 2233.94
  4971.1 2233.44  4986.2 2233.94  4995.4 2235.55  5020.0 2236.38  5028.4 2235.23
  5041.3 2235.57  5059.5 2238.87  5093.2 2238.78  5104.2 2243.24  5114.0 2249.29
  5133.3 2263.83  5138.5 2264.24  5145.1 2276.94  5155.5 2294.08  5172.8 2297.89
  5189.4 2297.61  5207.1 2297.87  5212.3 2296.22  5238.5 2296.43  5250.1 2294.67
#Mann=7,-1,0
  4540.6    0.07       0  4626.4    0.16       0  4876.0    0.07       0
  4970.6    0.07       0  4986.2    0.07       0  5028.4    0.16       0
  5189.4    0.07       0
Bank Sta=4970.6,4986.2
Exp/Cntr=0.3,0.1

Type RM Length L Ch R = 1,18036,273,273,273
BEGIN DESCRIPTION:
Little Elm Creek 2 18036.31
END DESCRIPTION:
XS GIS Cut Line= 3
      1501716.98      6766616.81      1502310.71      6766512.64
      1502567.96      6766452.88
#Sta/Elev= 30
  4401.3 2283.22  4447.3 2276.10  4478.3 2271.72  4531.3 2268.90  4561.7 2265.78
  4622.6 2256.16  4764.8 2251.41  4805.4 2244.08  4824.5 2242.02  4937.4 2241.17
  4951.8 2237.92  4967.8 2233.97  4988.1 2233.78  4997.6 2232.13  5001.1 2229.88
  5001.6 2229.38  5016.7 2229.88  5018.8 2233.12  5039.3 2245.55  5045.6 2251.99
  5050.7 2250.34  5068.9 2262.20  5080.4 2269.75  5088.2 2277.21  5093.3 2278.98
  5100.9 2288.85  5111.2 2295.37  5136.0 2299.91  5203.6 2306.91  5268.2 2308.22
#Mann=6,-1,0
  4401.3    0.07       0  4447.3    0.16       0  4951.8    0.07       0
  5001.1    0.07       0  5016.7    0.07       0  5068.9    0.16       0
Bank Sta=5001.1,5016.7
Exp/Cntr=0.3,0.1

Type RM Length L Ch R = 1,17763,185,185,185
BEGIN DESCRIPTION:
Little Elm Creek 2 17762.729
END DESCRIPTION:
XS GIS Cut Line= 3
      1501755.00      6766738.00      1502355.27      6766771.46
      1502554.98      6766738.00
#Sta/Elev= 30
  4398.8 2279.46  4438.9 2270.29  4478.9 2264.52  4549.0 2252.43  4579.1 2250.22
  4639.2 2248.91  4671.3 2246.10  4739.3 2244.05  4779.4 2238.79  4853.8 2238.59
  4869.5 2238.13  4891.8 2230.15  4892.3 2229.65  4907.4 2230.15  4909.6 2232.13
  4919.6 2233.87  4939.6 2234.42  4979.7 2231.58  5020.0 2232.14  5040.3 2241.36
  5048.3 2248.49  5053.4 2247.58  5070.7 2268.04  5080.8 2276.08  5109.0 2285.69
  5114.0 2285.84  5131.5 2290.30  5169.6 2297.22  5192.4 2299.19  5202.5 2301.40
#Mann=4,-1,0
  4398.8    0.16       0  4853.8    0.07       0  4891.8    0.07       0
  4907.4    0.07       0
Bank Sta=4891.8,4907.4
Exp/Cntr=0.3,0.1

Type RM Length L Ch R = 1,17578,155,155,155
BEGIN DESCRIPTION:
Little Elm Creek 2 17578.18
END DESCRIPTION:
XS GIS Cut Line= 3
      1501656.98      6766938.67      1502303.76      6766942.13
      1502651.56      6766890.47
#Sta/Elev= 30
  4347.0 2296.68  4375.0 2293.05  4393.7 2288.46  4415.0 2283.16  4455.0 2268.14
  4515.0 2253.80  4545.0 2249.10  4626.8 2243.73  4675.0 2242.12  4715.0 2236.52
  4853.4 2236.94  4865.0 2237.13  4875.0 2234.76  4885.0 2228.93  4895.0 2228.76
  4955.0 2233.97  4975.0 2231.37  4984.1 2227.64  4984.6 2227.14  4999.7 2227.64
  5025.4 2230.74  5035.5 2235.22  5052.2 2246.37  5058.3 2246.15  5086.0 2270.53
  5096.1 2274.30  5187.1 2283.81  5218.9 2289.68  5247.1 2293.39  5345.4 2307.11
#Mann=9,-1,0
  4347.0    0.07       0  4393.7    0.16       0  4626.8    0.12       0
  4853.4    0.07       0  4984.1    0.07       0  4999.7    0.07       0
  5052.2   0.035       0  5218.9    0.16       0  5247.1   0.035       0
Bank Sta=4984.1,4999.7
Exp/Cntr=0.3,0.1

Type RM Length L Ch R = 1,17423,246,246,246
BEGIN DESCRIPTION:
Little Elm Creek 2 17422.64
END DESCRIPTION:
XS GIS Cut Line= 3
      1501691.59      6767097.77      1502272.63      6767080.47
      1502700.70      6767049.40
#Sta/Elev= 30
  4435.3 2290.86  4458.7 2288.37  4488.7 2282.67  4528.8 2270.71  4578.8 2258.59
  4594.7 2252.59  4605.9 2250.91  4637.0 2244.98  4678.8 2238.34  4718.8 2235.49
  4801.1 2235.24  4890.8 2236.11  4918.9 2236.25  4938.9 2234.14  4991.2 2225.27
  4991.7 2224.77  5006.8 2225.27  5049.1 2229.24  5079.1 2253.18  5089.2 2257.77
  5101.7 2260.45  5117.0 2265.35  5139.3 2270.02  5199.5 2274.15  5219.5 2272.88
  5256.3 2274.96  5269.6 2279.58  5279.3 2281.32  5359.9 2296.13  5445.8 2307.90
#Mann=9,-1,0
  4435.3    0.07       0  4605.9    0.16       0  4637.0    0.12       0
  4801.1    0.16       0  4890.8    0.07       0  4991.2    0.07       0
  5006.8    0.07       0  5101.7   0.035       0  5279.3    0.16       0
Bank Sta=4991.2,5006.8
Exp/Cntr=0.3,0.1

Type RM Length L Ch R = 1,17177,239,239,239
BEGIN DESCRIPTION:
Little Elm Creek 2 17176.84
END DESCRIPTION:
XS GIS Cut Line= 3
      1501663.91      6767274.16      1502200.00      6767312.20
      1502767.19      6767198.07
#Sta/Elev= 30
  4457.4 2279.36  4497.7 2277.83  4528.7 2276.25  4588.8 2265.88  4669.0 2261.42
  4689.1 2254.91  4699.1 2247.39  4718.8 2235.89  4723.9 2236.44  4729.2 2233.26
  4859.5 2233.28  4907.1 2231.55  4959.8 2230.65  4979.8 2227.86  4982.0 2224.65
  4982.5 2224.15  4997.6 2224.65  5043.7 2224.70  5081.5 2240.88  5089.4 2241.95
  5149.5 2242.00  5191.1 2240.71  5285.6 2247.78  5336.6 2248.84  5346.2 2251.28
  5387.6 2263.60  5408.0 2276.12  5445.3 2293.89  5496.2 2303.80  5573.4 2311.68
#Mann=7,-1,0
  4457.4    0.07       0  4497.7    0.16       0  4907.1    0.07       0
  4982.0    0.07       0  4997.6    0.07       0  5149.5   0.035       0
  5346.2    0.16       0
Bank Sta=4982,4997.6
Exp/Cntr=0.3,0.1

Type RM Length L Ch R = 1,16938,191,191,191
BEGIN DESCRIPTION:
Little Elm Creek 2 16937.69
END DESCRIPTION:
XS GIS Cut Line= 3
      1501670.85      6767609.65      1502161.95      6767533.56
      1502851.87      6767309.34
#Sta/Elev= 30
  4510.8 2275.05  4596.0 2270.81  4717.4 2258.85  4737.6 2250.27  4746.4 2238.72
  4751.5 2237.10  4757.9 2230.08  4768.0 2227.01  4923.5 2227.32  4960.2 2227.95
  4970.4 2226.93  4982.8 2222.61  4983.3 2222.11  4998.4 2222.61  5021.5 2224.30
  5053.0 2223.28  5063.5 2227.48  5071.5 2233.14  5116.1 2230.44  5172.6 2237.70
  5201.5 2238.68  5294.9 2237.41  5419.2 2240.44  5497.4 2243.84  5515.7 2247.35
  5547.2 2259.03  5610.3 2291.46  5631.3 2297.21  5662.9 2301.48  5733.2 2304.68
#Mann=6,-1,0
  4510.8    0.16       0  4923.5    0.07       0  4982.8    0.07       0
  4998.4    0.07       0  5201.5   0.035       0  5419.2    0.16       0
Bank Sta=4982.8,4998.4
Exp/Cntr=0.3,0.1

Type RM Length L Ch R = 1,16747,330,330,330
BEGIN DESCRIPTION:
Little Elm Creek 2 16746.66
END DESCRIPTION:
XS GIS Cut Line= 3
      1501643.11      6767734.16      1502106.61      6767709.95
      1502921.46      6767585.65
#Sta/Elev= 30
  4537.9 2276.96  4660.0 2269.80  4748.5 2259.28  4810.2 2254.62  4830.2 2249.55
  4870.2 2226.60  4890.3 2224.43  4952.9 2225.78  5002.0 2224.51  5002.7 2219.61
  5003.2 2219.11  5018.3 2219.61  5030.7 2221.79  5061.1 2222.21  5091.4 2231.37
  5102.8 2231.39  5274.7 2230.22  5334.2 2233.85  5374.7 2231.42  5384.8 2233.84
  5466.5 2237.44  5575.3 2241.57  5597.2 2244.24  5637.7 2243.83  5678.1 2255.77
  5698.4 2266.01  5718.6 2279.62  5746.5 2292.14  5775.9 2298.69  5826.3 2302.89
#Mann=8,-1,0
  4537.9    0.16       0  4952.9    0.07       0  5002.7    0.07       0
  5018.3    0.07       0  5102.8    0.16       0  5274.7   0.035       0
  5466.5    0.16       0  5746.5    0.07       0
Bank Sta=5002.7,5018.3
Exp/Cntr=0.3,0.1

Type RM Length L Ch R = 1,16417,195,195,195
BEGIN DESCRIPTION:
Little Elm Creek 2 16417.27
END DESCRIPTION:
XS GIS Cut Line= 3
      1501719.21      6768010.86      1502200.00      6768010.86
      1502950.28      6767620.15
#Sta/Elev= 30
  4513.9 2270.96  4769.7 2260.96  4779.7 2259.18  4819.7 2234.32  4839.7 2225.24
  4859.7 2221.59  4897.4 2222.44  4911.8 2217.37  4912.3 2216.87  4927.5 2217.37
  4929.7 2220.15  4949.7 2221.27  4994.7 2218.22  5022.9 2227.08  5065.1 2227.73
  5279.8 2226.93  5442.7 2229.04  5572.2 2232.93  5616.4 2237.24  5676.8 2246.75
  5699.1 2256.01  5711.5 2264.31  5733.2 2277.23  5743.3 2281.02  5749.0 2286.43
  5765.4 2291.63  5771.1 2296.66  5787.5 2295.47  5793.2 2298.92  5840.6 2305.01
#Mann=8,-1,0
  4513.9    0.16       0  4897.4    0.07       0  4911.8    0.07       0
  4927.5    0.07       0  5065.1    0.16       0  5279.8   0.035       0
  5442.7    0.16       0  5711.5    0.07       0
Bank Sta=4911.8,4927.5
Exp/Cntr=0.3,0.1

Type RM Length L Ch R = 1,16222,365,365,365
BEGIN DESCRIPTION:
Little Elm Creek 2 16221.93
END DESCRIPTION:
XS GIS Cut Line= 3
      1501698.48      6768360.18      1502279.55      6768166.50
      1502969.32      6767752.63
#Sta/Elev= 30
  4384.0 2270.06  4414.7 2268.81  4429.4 2267.97  4464.7 2266.10  4506.8 2258.15
  4612.2 2252.60  4633.3 2256.84  4812.5 2255.81  4849.7 2231.21  4875.8 2218.87
  4973.3 2215.96  4973.8 2215.46  4989.0 2215.96  5017.7 2225.45  5239.6 2225.81
  5424.2 2225.06  5546.3 2225.43  5610.5 2231.80  5626.0 2236.47  5641.6 2247.27
  5647.4 2246.81  5662.9 2259.84  5684.3 2267.21  5699.9 2282.19  5705.7 2281.45
  5721.3 2298.75  5727.1 2296.78  5736.8 2302.26  5756.8 2304.99  5800.9 2305.53
#Mann=10,-1,0
  4384.0   0.035       0  4414.7    0.07       0  4429.4    0.16       0
  4849.7    0.07       0  4973.3    0.07       0  4989.0    0.07       0
  5017.7    0.16       0  5239.6   0.035       0  5424.2    0.16       0
  5756.8    0.07       0
Bank Sta=4973.3,4989
Exp/Cntr=0.3,0.1

Type RM Length L Ch R = 1,15857,232,232,232
BEGIN DESCRIPTION:
Little Elm Creek 2 15856.67
END DESCRIPTION:
XS GIS Cut Line= 3
      1501968.25      6768678.39      1502417.89      6768457.02
      1502915.95      6767803.32
#Sta/Elev= 30
  4495.6 2260.47  4548.7 2258.71  4685.8 2249.19  4845.2 2251.36  4918.2 2232.55
  4957.6 2228.51  4971.3 2215.29  4993.1 2210.86  4993.6 2210.36  5008.9 2210.86
  5065.5 2214.49  5086.3 2222.19  5128.9 2213.78  5157.5 2222.04  5433.7 2223.38
  5643.4 2225.20  5672.5 2235.08  5693.3 2249.02  5707.8 2250.49  5722.4 2259.07
  5728.6 2266.97  5736.9 2267.36  5743.2 2275.13  5757.7 2275.53  5764.0 2283.16
  5772.2 2283.50  5778.5 2296.02  5786.8 2292.13  5793.1 2299.78  5818.6 2305.27
#Mann=8,-1,0
  4495.6    0.07       0  4548.7   0.035       0  4685.8    0.07       0
  4993.1    0.07       0  5008.9    0.07       0  5128.9    0.16       0
  5157.5   0.035       0  5433.7    0.16       0
Bank Sta=4993.1,5008.9
Exp/Cntr=0.3,0.1

Type RM Length L Ch R = 1,15625,170,170,170
BEGIN DESCRIPTION:
Little Elm Creek 2 15624.7
END DESCRIPTION:
XS GIS Cut Line= 3
      1502030.56      6768757.91      1502628.87      6768519.28
      1503070.81      6767970.31
#Sta/Elev= 30
  4350.2 2257.91  4354.6 2257.91  4430.3 2255.28  4484.2 2248.41  4520.5 2240.16
  4538.0 2241.99  4559.5 2249.45  4613.4 2249.87  4636.8 2248.72  4661.1 2241.68
  4685.4 2230.85  4839.9 2227.02  4893.3 2225.04  4930.6 2214.57  5013.7 2210.47
  5014.2 2209.97  5029.5 2210.47  5034.5 2213.48  5085.6 2212.44  5127.3 2214.43
  5132.6 2217.36  5184.8 2220.25  5291.3 2218.07  5341.6 2222.61  5362.4 2230.96
  5405.6 2240.39  5476.0 2285.82  5483.8 2294.59  5525.7 2296.54  5699.1 2311.54
#Mann=8,-1,0
  4350.2    0.16       0  4354.6   0.035       0  4520.5    0.07       0
  4839.9   0.035       0  5013.7   0.035       0  5029.5   0.035       0
  5132.6    0.16       0  5525.7    0.07       0
Bank Sta=5013.7,5029.5
Exp/Cntr=0.3,0.1

Type RM Length L Ch R = 1,15455,234,234,234
BEGIN DESCRIPTION:
Little Elm Creek 2 15455.34
END DESCRIPTION:
XS GIS Cut Line= 3
      1502054.71      6768861.70      1502781.05      6768571.16
      1503196.12      6768235.65
#Sta/Elev= 30
  4213.1 2253.83  4268.0 2256.14  4330.2 2249.22  4370.4 2238.47  4375.7 2240.48
  4394.6 2236.66  4400.0 2239.30  4424.2 2231.89  4478.1 2227.76  4885.2 2220.53
  4962.7 2220.03  4968.1 2216.12  4987.0 2214.86  4992.3 2208.70  4999.7 2207.93
  5000.2 2207.43  5015.6 2207.93  5135.6 2215.54  5199.5 2215.32  5220.3 2223.45
  5257.0 2251.17  5263.5 2253.13  5270.5 2259.99  5277.9 2277.32  5284.3 2274.18
  5292.2 2292.43  5298.3 2289.65  5306.6 2298.15  5434.5 2309.75  5529.1 2313.20
#Mann=6,-1,0
  4213.1    0.16       0  4330.2   0.035       0  4885.2    0.16       0
  4999.7    0.07       0  5015.6    0.16       0  5298.3    0.07       0
Bank Sta=4999.7,5015.6
Exp/Cntr=0.3,0.1
