HEC-RAS study Lytle Creek.prj: Lytle Creek Base Level Engineering

--- Lytle Creek.g01 (geometry) --- (continued)

Type RM Length L Ch R = 1 ,32322   ,366,366,366
BEGIN DESCRIPTION:
Lytle Creek 32322.286
END DESCRIPTION:
XS GIS Cut Line= 3
      1600844.22      6825531.33      1601848.88      6825540.18
      1603549.03      6826020.91
#Sta/Elev= 30
  3995.3 1759.99  4326.1 1758.03  4536.1 1760.18  4746.1 1758.67  4826.1 1754.74
  4906.1 1748.86  4946.1 1744.65  4966.1 1742.35  4973.5 1733.41  4974.6 1732.81
  5026.5 1733.41  5050.1 1735.19  5068.7 1741.79  5123.5 1743.06  5235.5 1741.57
  5264.3 1742.14  5276.5 1740.12  5303.5 1739.86  5342.6 1734.61  5370.1 1737.23
  5381.8 1740.37  5401.3 1742.19  5512.6 1741.94  6000.7 1742.26  6005.9 1743.02
  6366.4 1744.77  6512.6 1748.12  6664.1 1753.45  6703.2 1755.82  6766.8 1756.41
#Mann= 5 ,-1 , 0
  3995.3     .05       0  4973.5     .05       0  5026.5     .05       0
  5123.5     .12       0  5512.6     .05       0
Bank Sta=4973.5,5026.5
XS Rating Curve= 0 ,0
Exp/Cntr=0.3,0.1

Type RM Length L Ch R = 1 ,31956   ,530,530,530
BEGIN DESCRIPTION:
Lytle Creek 31167.796
END DESCRIPTION:
XS GIS Cut Line= 3
      1600882.34      6825770.91      1602250.42      6825916.75
      1603524.75      6826309.11
#Sta/Elev= 30
  4093.9 1760.14  4327.9  1759.4  4682.3  1753.4  4850.8 1753.02  4911.2 1748.74
  4921.2 1746.69  4951.4 1733.92  4971.5 1733.85  4973.5 1732.05  4974.6 1731.45
  5026.5 1732.05  5031.8 1738.76  5041.9 1739.48    5052  1739.4    5057 1736.89
  5092.2 1736.49  5132.4 1742.04  5162.6 1742.65  5189.6 1740.49  5212.9 1736.44
  5222.9 1732.53  5241.9 1735.79  5246.9 1734.77  5253.1 1739.68  5263.1 1741.31
  5577.3 1740.63    5692 1740.21  6344.4  1747.1  6667.3 1756.18  6803.1 1757.11
#Mann= 5 ,-1 , 0
  4093.9     .05       0  4973.5     .05       0  5026.5     .05       0
  5189.6     .12       0  5577.3     .05       0
Bank Sta=4973.5,5026.5
XS Rating Curve= 0 ,0
Exp/Cntr=0.3,0.1

Type RM Length L Ch R = 1 ,31426   ,172,172,172
BEGIN DESCRIPTION:
Mapping XS 7648e034
END DESCRIPTION:
XS GIS Cut Line= 3
      1600986.55      6826121.61      1602861.54      6826319.52
       1603500.2      6826357.71
#Sta/Elev= 30
  3875.4 1758.96  3914.1 1757.35  3934.2 1758.73  4004.6 1753.76  4044.8 1753.12
    4085 1750.28  4155.4 1749.37  4225.8 1746.35  4456.1 1742.79  4842.7 1741.62
  4899.5 1740.19  4935.6 1735.86  4969.9 1733.92  4971.7 1730.35    4973 1729.55
  5028.3 1730.35  5033.5 1730.74  5050.3 1736.48  5060.4  1738.5  5080.5  1739.6
  5120.7 1740.13  5241.4 1736.54  5291.7 1738.94  5410.1 1740.42  5462.6 1743.15
  5924.6 1746.73  6074.8 1749.77  6275.2 1756.45  6385.4 1758.34  6400.6 1757.33
#Mann= 3 ,-1 , 0
  3875.4     .05       0  4971.7     .05       0  5028.3     .05       0
Bank Sta=4971.7,5028.3
XS Rating Curve= 0 ,0
Exp/Cntr=0.3,0.1

Type RM Length L Ch R = 1 ,31254   ,650,650,650
BEGIN DESCRIPTION:
Mapping XS e18eeca7
END DESCRIPTION:
XS GIS Cut Line= 4
      1601538.66       6826298.7      1601764.31      6826326.47
      1602802.51      6826583.41      1603461.16      6826694.34
#Sta/Elev= 30
  4440.4 1754.75  4446.8 1753.99  4473.8 1743.38  4497.2 1741.99    4729 1741.06
  4817.7 1741.39  4874.5 1741.12    4926 1739.41  4936.3 1734.83  4943.1 1733.55
  4948.2 1733.22  4967.2 1735.72  4971.7 1727.96    4973 1727.16    5027 1727.16
  5028.3 1727.96  5031.1 1738.75  5059.9 1741.96    5266  1738.8  5279.5 1737.91
  5286.6 1735.03  5307.2 1733.27  5338.1 1737.77  5502.9 1743.97  5911.3 1746.53
  5993.3 1748.28  6165.7  1755.1  6226.6  1756.4    6335 1757.13  6405.2 1756.15
#Mann= 5 ,-1 , 0
  4440.4     .05       0    4729     .12       0  4817.7     .05       0
  4971.7     .05       0  5028.3     .05       0
Bank Sta=4971.7,5028.3
XS Rating Curve= 0 ,0
Exp/Cntr=0.3,0.1

Type RM Length L Ch R = 1 ,30604   ,411,411,411
BEGIN DESCRIPTION:
Mapping XS 778433d1
END DESCRIPTION:
XS GIS Cut Line= 2
      1601437.97      6826961.89      1603246.96      6827038.27
#Sta/Elev= 30
  4582.7 1750.48  4589.7 1754.24  4599.7  1754.5  4611.9 1751.58  4629.8 1742.85
  4639.8 1740.12  4659.8 1738.42  4709.8 1738.74  4719.8 1741.06  4739.9 1738.78
  4904.3 1740.85  4950.1 1737.29  4970.1 1730.55  4971.7 1726.66    4973 1725.86
  5028.3 1726.66  5030.1 1738.97  5079.1  1740.5  5204.1 1739.83  5271.4 1739.33
  5291.3 1739.41  5400.5 1737.81  5440.5  1734.5  5470.5 1739.43  5500.5 1732.46
  5510.6 1732.16  5670.7 1748.95  5760.8 1748.36  6231.2 1756.35  6393.3 1756.23
#Mann= 7 ,-1 , 0
  4582.7     .05       0  4904.3     .12       0  4971.7     .07       0
  5028.3     .12       0  5204.1     .05       0  5271.4     .12       0
  5291.3     .05       0
Bank Sta=4971.7,5028.3
XS Rating Curve= 0 ,0
Exp/Cntr=0.3,0.1

Type RM Length L Ch R = 1 ,30193   ,605,605,605
BEGIN DESCRIPTION:
Mapping XS 8268765c
END DESCRIPTION:
XS GIS Cut Line= 3
      1601413.63      6827177.17      1602115.01      6827531.33
      1603726.14      6827694.53
#Sta/Elev= 30
  4588.2 1752.02  4598.2 1753.92  4612.1 1753.39  4620.5 1748.71  4626.1 1748.17
  4642.8 1740.58  4665.1 1738.25  4823.7 1739.46  4828.9 1739.56  4932.1 1739.44
  4938.3 1738.62  4948.2 1734.06    4955 1726.66  4971.7 1725.99    4973 1725.19
  5028.3 1725.99  5037.8 1732.06  5044.1 1733.91  5080.1 1733.42  5094.3 1734.11
    5111 1739.98  5119.5 1739.94  5309.8 1738.11  5424.2    1739  5489.6 1736.72
  5524.7 1738.08  5544.8 1734.51  5715.7 1738.58  6358.9 1744.24  6993.3 1757.54
#Mann= 9 ,-1 , 0
  4588.2     .05       0  4823.7     .12       0  4828.9     .05       0
  4932.1     .12       0  4971.7     .07       0  5028.3     .12       0
  5080.1     .05       0  5119.5     .12       0  5309.8     .05       0
Bank Sta=4971.7,5028.3
XS Rating Curve= 0 ,0
Exp/Cntr=0.3,0.1

Type RM Length L Ch R = 1 ,29588   ,1049,1049,1049
BEGIN DESCRIPTION:
Mapping XS cfcc106c
END DESCRIPTION:
XS GIS Cut Line= 3
      1601326.81        6827698.       1602441.4      6827906.33
       1603746.9       6828034.8
#Sta/Elev= 30
  4362.3 1751.27  4370.6 1753.82  4387.7 1752.47  4421.5  1740.7  4440.4 1737.37
  4750.5 1739.28  4787.7 1741.55  4797.9 1740.06  4824.1 1729.49  4848.8 1732.15
  4858.5 1735.91  4869.1 1738.81  4881.9 1738.61  4899.6 1733.45    4920 1731.88
  4960.7 1734.42  4970.8 1728.07  4971.7 1724.25    4973 1723.45  5028.3 1724.25
  5031.9  1736.1  5034.3 1736.93  5039.8 1738.83  5199.4 1737.62  5296.4 1737.69
  5326.9 1734.94  5365.9 1738.52  5610.3 1738.91    6163 1744.76    6808 1758.38
#Mann= 7 ,-1 , 0
  4362.3     .05       0  4750.5     .12       0  4858.5     .05       0
  4971.7     .05       0  5028.3     .05       0  5034.3     .12       0
  5199.4     .05       0
Bank Sta=4971.7,5028.3
XS Rating Curve= 0 ,0
Exp/Cntr=0.3,0.1

Type RM Length L Ch R = 1 ,28539   ,663,663,663
BEGIN DESCRIPTION:
Mapping XS 4e40e666
END DESCRIPTION:
XS GIS Cut Line= 3
      1601212.22      6828263.97       1601753.9      6828475.77
      1603257.41      6828982.73
#Sta/Elev= 30
  4798.9 1754.17  4820.8 1752.13  4844.8 1743.84  4850.7 1740.04  4866.3 1737.56
  4910.4 1737.44  4964.7 1732.58  4971.7 1720.71    4973 1719.91  5028.3 1720.71
  5038.1 1731.86  5043.4 1736.03  5048.8 1737.63    5101 1736.83  5374.6 1736.74
  5413.3 1736.01  5431.8  1732.3    5445 1731.67  5463.3 1735.17  5519.3 1735.83
  5622.8 1735.16    5841 1736.08  5850.3 1734.89  5867.1 1733.93  5877.8 1736.31
  6056.1 1738.13  6155.8 1743.69  6344.7 1749.09  6616.4 1753.42  6967.2 1755.63
#Mann= 7 ,-1 , 0
  4798.9     .05       0  4971.7     .03       0  5028.3     .05       0
    5101     .12       0  5519.3     .05       0  5622.8     .12       0
  5850.3     .05       0
Bank Sta=4971.7,5028.3
XS Rating Curve= 0 ,0
Exp/Cntr=0.3,0.1

Type RM Length L Ch R = 1 ,27876   ,688,688,688
BEGIN DESCRIPTION:
Lytle Creek 27783.321
END DESCRIPTION:
XS GIS Cut Line= 3
      1599414.49      6828785.67       1601862.4      6828889.84
      1602586.33      6829285.65
#Sta/Elev= 30
  2760.1 1748.54  2934.1 1742.68  2980.8 1738.47  3070.9 1733.45  3110.9 1731.52
    3201 1730.35    3241 1728.56  3261.1 1725.59  3281.1 1730.36  3342.7 1731.73
  3591.4 1732.06  3733.3 1730.62  3951.7 1730.06  4181.9 1733.03  4511.2 1733.82
  4717.1 1734.89  4835.3 1735.77  4902.5 1735.21  4918.5 1733.58  4952.6 1729.46
  4962.6    1727  4971.6 1721.28  4972.9 1720.48  5028.5 1721.28  5032.7 1733.81
  5042.7 1739.57  5092.7  1741.8    5566 1751.03  5828.6 1748.63  6035.3 1748.94
#Mann= 9 ,-1 , 0
  2760.1     .05       0  3342.7     .12       0  3733.3     .05       0
  4511.2     .12       0  4717.1     .05       0  4835.3     .12       0
  4918.5     .05       0  4971.6     .05       0  5028.5     .05       0
Bank Sta=4971.6,5028.5
XS Rating Curve= 0 ,0
Exp/Cntr=0.3,0.1

Type RM Length L Ch R = 1 ,27188   ,907,907,907
BEGIN DESCRIPTION:
Lytle Creek 27188.48
END DESCRIPTION:
XS GIS Cut Line= 3
      1599216.53      6829051.29      1601206.35      6829336.08
       1602086.4      6829842.98
#Sta/Elev= 30
  2989.9 1750.79  3382.3 1733.22  3503.6 1730.69  3715.7 1730.66  3806.6 1726.54
  3816.7 1724.52  3921.2 1725.54    3948 1730.44  4198.7 1728.37    4241 1724.87
  4281.4 1728.48  4372.3 1730.39  4916.1 1734.58  4964.7    1735  4968.3 1735.06
  4971.6 1721.23  4972.9 1720.43  5028.5 1721.23  5030.6 1723.04  5052.2 1721.82
  5067.7 1731.72  5079.5 1734.52  5187.9 1733.48  5277.7 1732.53  5363.8 1734.75
  5432.9 1739.91  5609.6 1746.11  5674.3 1747.37  5806.3 1745.21  6015.6 1748.44
#Mann= 7 ,-1 , 0
  2989.9     .05       0  4916.1     .12       0  4964.7     .05       0
  4971.6     .05       0  5028.5     .05       0  5187.9     .12       0
  5363.8     .05       0
Bank Sta=4971.6,5028.5
XS Rating Curve= 0 ,0
Exp/Cntr=0.3,0.1

Type RM Length L Ch R = 1 ,26281   ,1679,1679,1679
BEGIN DESCRIPTION:
Lytle Creek 26661.68
END DESCRIPTION:
XS GIS Cut Line= 3
      1598860.62      6829910.67      1601027.33      6829917.61
      1601732.22      6830153.73
#Sta/Elev= 30
  3205.6 1748.66    3280 1747.11    3440 1738.67    3520 1732.52    3610 1729.82
    3690 1729.08    4380 1727.39    4420 1723.65    4440 1726.12    4470 1727.19
    4530 1726.78    4570 1724.01    4600 1725.96    4760 1728.58    4850 1732.41
    4930 1733.75    4940 1732.63    4960 1721.48  4971.6 1719.33  4972.9 1718.53
  5028.5 1719.33    5030 1733.27  5475.3 1730.78  5576.8    1732  5591.3 1731.47
    5623 1726.25  5645.2 1731.83  5760.1 1735.46    5909 1742.41  6115.7 1749.75
#Mann= 4 ,-1 , 0
  3205.6     .05       0  4971.6     .05       0  5028.5     .05       0
    5909     .05       0
Bank Sta=4971.6,5028.5
XS Rating Curve= 0 ,0
Exp/Cntr=0.3,0.1

Type RM Length L Ch R = 1 ,24602   ,364,364,364
BEGIN DESCRIPTION:
Lytle Creek 24387.649
END DESCRIPTION:
XS GIS Cut Line= 3
      1598867.58      6830452.33      1601270.39      6830709.28
      1601624.59      6830559.96
#Sta/Elev= 30
    3101 1749.19  3148.7 1749.82  3188.9 1746.65  3319.7 1741.94  3621.4 1727.13
    3903 1724.99  4048.3 1726.19  4104.1 1725.22  4134.3 1720.86  4154.4 1723.71
  4427.4 1728.48  4466.2 1727.78  4486.3 1729.37  4938.8 1730.97  4948.9 1730.78
    4959 1727.79    4969 1721.93  4971.5 1715.44  4972.8 1714.64  5028.5 1715.44
  5029.4 1726.01  5059.5 1730.25  5089.3 1729.72  5230.5 1731.24    5324 1735.28
  5365.3 1735.84  5457.6 1740.89  5589.1 1741.41  5620.2 1745.72  5901.9 1747.11
#Mann= 5 ,-1 , 0
    3101     .05       0  4971.5     .05       0  5028.5     .05       0
  5089.3     .12       0    5324     .05       0
Bank Sta=4971.5,5028.5
XS Rating Curve= 0 ,0
Exp/Cntr=0.3,0.1

Type RM Length L Ch R = 1 ,24238   ,477,477,477
BEGIN DESCRIPTION:
Lytle Creek 23884.878
END DESCRIPTION:
XS GIS Cut Line= 3
      1599058.61      6830910.67      1601180.11      6831018.31
      1601443.97      6830869.02
#Sta/Elev= 30
  3238.6 1743.52  3315.1 1743.64  3395.2 1741.27  3475.3 1737.18  3595.4 1729.19
  3645.5 1727.14  3685.6 1723.85  3715.6 1722.85  3805.7 1724.44  3845.8 1724.04
  3865.8 1722.81  3878.7 1719.63  3885.8 1721.13  3915.9 1723.12  4226.3 1726.83
  4756.9 1728.64  4857.1 1729.98  4907.1 1729.05  4957.2 1729.53  4967.2 1726.59
  4971.5 1715.68  4972.8 1714.88  5027.2 1714.88  5028.5 1715.68  5037.3 1726.05
  5047.3 1730.01  5368.2 1729.62  5476.4  1733.9  5541.3 1738.93    5666 1743.83
#Mann= 3 ,-1 , 0
  3238.6     .05       0  4971.5     .05       0  5028.5     .05       0
Bank Sta=4971.5,5028.5
XS Rating Curve= 0 ,0
Exp/Cntr=0.3,0.1

Type RM Length L Ch R = 1 ,23761   ,544,544,544
BEGIN DESCRIPTION:
Lytle Creek 23335.647
END DESCRIPTION:
XS GIS Cut Line= 3
       1599093.3      6831039.14       1600881.5      6831372.48
      1601975.23      6831737.05
#Sta/Elev= 30
  3051.6 1741.27  3195.7 1739.25  3266.9 1731.92  3512.7 1723.46    3745 1724.85
  3867.1 1719.25  3877.3 1719.51  3886.8 1723.33  3989.2 1726.52  4192.6 1724.14
  4284.2 1728.91  4375.7 1726.22  4497.8 1729.04  4823.6 1726.91  4853.8 1728.98
  4970.8 1722.82  4971.2  1716.8  4972.6    1716  5028.8  1716.8    5034 1728.34
  5060.4  1729.3  5160.5 1728.89  5192.1 1722.69  5218.5 1727.84  5223.8 1725.18
  5295.9 1727.86  5359.2 1724.52  5408.2 1728.62    5540 1729.34  6023.5 1745.73
#Mann= 3 ,-1 , 0
  3051.6     .05       0  4971.2     .05       0  5028.8     .05       0
Bank Sta=4971.2,5028.8
XS Rating Curve= 0 ,0
Exp/Cntr=0.3,0.1

Type RM Length L Ch R = 1 ,23217   ,414,414,414
BEGIN DESCRIPTION:
Lytle Creek 22765.807
END DESCRIPTION:
XS GIS Cut Line= 3
      1599135.01      6831181.52      1600853.72      6831820.39
      1602050.84       6832431.1
#Sta/Elev= 30
  3274.7 1743.09  3488.1 1736.38  3713.4 1722.44  3879.6 1724.73  3940.3  1718.3
  4042.8 1724.48  4308.2  1725.9  4405.5 1717.36  4626.1  1718.6  4693.6 1726.43
  4797.5 1728.69    4969 1722.64  4971.2 1714.46  4972.6 1713.66  5028.8 1714.46
  5029.7 1728.01    5085 1730.95  5181.4 1729.87  5225.8 1724.09  5278.1    1728
  5292.5 1724.12    5537 1730.36  5709.3 1743.53    5776 1742.08  5859.3 1749.85
  5909.3 1762.88  5985.4 1770.93  6410.9 1770.52  6442.9 1770.73  6452.2    1771
#Mann= 5 ,-1 , 0
  3274.7     .05       0  4971.2     .03       0  5028.8     .05       0
  6410.9     .12       0  6442.9     .05       0
Bank Sta=4971.2,5028.8
XS Rating Curve= 0 ,0
Exp/Cntr=0.3,0.1

Type RM Length L Ch R = 1 ,22803   ,2734,2734,2734
BEGIN DESCRIPTION:
Lytle Creek 22183.167
END DESCRIPTION:
XS GIS Cut Line= 3
      1599242.59      6831684.97       1600919.7      6832250.95
       1602169.7      6832816.92
#Sta/Elev= 30
  3562.3 1739.13  3652.3 1739.46  3786.5 1734.75  3849.8 1729.95  3898.7 1717.75
  3961.7 1723.09  4092.8 1722.02  4208.1 1727.16  4324.7 1724.14  4968.6 1728.34
  4971.2  1714.5  4972.6  1713.7  5028.8  1714.5  5031.9 1718.95  5052.5 1724.64
  5120.7 1726.94  5316.8 1723.04    5393 1730.85  5502.2 1734.32  5546.7  1740.8
  5726.5 1747.26  5766.3 1751.46    5842 1749.94  6073.6 1756.17  6112.6 1760.52
  6279.8 1761.28  6331.5 1755.86  6423.9 1761.19  6579.6 1762.15  6704.5 1765.35
#Mann= 4 ,-1 , 0
  3562.3     .05       0  4971.2     .03       0  5028.8     .05       0
  6579.6     .12       0
Bank Sta=4971.2,5028.8
XS Rating Curve= 0 ,0
Exp/Cntr=0.3,0.1

Type RM Length L Ch R = 1 ,20069   ,623,623,623
BEGIN DESCRIPTION:
Mapping XS ea394c71
END DESCRIPTION:
XS GIS Cut Line= 3
      1599106.33      6831910.67      1600204.42      6832978.38
      1600902.64      6833533.49
#Sta/Elev= 30
  4380.3 1744.43  4511.8 1747.46    4731 1737.42  4773.5 1734.58  4823.1 1726.01
  4893.8 1722.39  4964.3 1721.33  4969.5 1711.43    4971 1710.43  5030.6 1711.43
  5035.1 1721.04  5123.7 1723.47  5261.4 1722.08  5671.6 1725.65  5862.5  1725.5
  5954.4 1727.46  5983.3 1730.56  6047.3 1731.03  6111.4 1735.34  6154.7 1731.72
  6181.9  1726.8  6225.1  1726.1  6417.4 1732.26  6531.1 1750.96  6580.7 1756.17
  6652.9 1758.29  6716.9  1763.3  6730.3 1761.09  6752.2 1762.87  6803.9 1762.81
#Mann= 4 ,-1 , 0
  4380.3     .05       0  4969.5     .03       0  5030.6     .05       0
  5123.7     .05       0
Bank Sta=4969.5,5030.6
XS Rating Curve= 0 ,0
Exp/Cntr=0.3,0.1

Type RM Length L Ch R = 1 ,19446   ,630,630,630
BEGIN DESCRIPTION:
Mapping XS 5db95189
END DESCRIPTION:
XS GIS Cut Line= 4
      1598871.95      6832609.45      1599991.74      6833086.89
       1600191.4      6833186.71      1600660.09      6833677.11
#Sta/Elev= 30
  4304.5 1742.99  4383.9  1739.3  4442.4 1739.81    4466 1736.49    4495 1738.88
  4525.2 1734.79  4601.3 1734.43  4677.4 1727.94  4700.3 1727.74  4718.5 1730.32
  4747.5 1728.86  4771.2 1730.22  4852.9 1723.21  4960.1 1720.06  4969.5 1710.52
    4971 1709.52  5030.6 1710.52  5036.2  1721.3  5058.2 1722.35  5134.5 1721.16
  5439.6 1724.06  5628.3 1722.14  5645.1 1724.46  5689.8 1724.65  5783.9 1722.23
  5875.8 1726.09  5974.8 1734.39  6059.8 1749.04  6335.6 1759.03  6423.4 1760.15
#Mann= 3 ,-1 , 0
  4304.5     .05       0  4969.5     .03       0  5030.6     .05       0
Bank Sta=4969.5,5030.6
XS Rating Curve= 0 ,0
Exp/Cntr=0.3,0.1

Type RM Length L Ch R = 1 ,18816   ,413,413,413
BEGIN DESCRIPTION:
Mapping XS 94faf59f
END DESCRIPTION:
XS GIS Cut Line= 3
      1598633.21      6832978.36       1599544.7      6833664.14
      1600680.93      6833950.37
#Sta/Elev= 30
  4405.6 1742.99  4499.1 1741.33  4534.5 1738.52  4557.4 1739.63  4563.6 1737.31
  4581.1 1736.86  4599.3 1734.55  4678.2 1731.48    4799 1723.22  4934.3  1720.7
  4957.2  1715.3  4969.5 1710.12    4971 1709.12  5030.6 1710.12  5034.3 1720.32
  5057.2 1721.56  5513.2 1720.25  5722.1 1722.42  5885.1 1723.88  5911.3 1722.68
  5917.8 1720.73  5931.9  1721.7  6034.6 1726.77  6070.6 1734.38  6075.7 1733.03
  6111.7 1740.59  6116.8  1739.6  6152.7 1752.12  6399.3 1759.09    6718 1761.76
#Mann= 8 ,-1 , 0
  4405.6      .1       0  4581.1     .05       0  4599.3     .12       0
  4969.5     .07       0  5030.6     .12       0  5722.1     .05       0
  5885.1     .12       0  5931.9     .05       0
Bank Sta=4969.5,5030.6
XS Rating Curve= 0 ,0
Exp/Cntr=0.3,0.1

Type RM Length L Ch R = 1 ,18403   ,493,493,493
BEGIN DESCRIPTION:
Mapping XS 08cbe365
END DESCRIPTION:
XS GIS Cut Line= 4
       1598127.2      6833257.05       1598590.7      6833538.27
      1599783.41      6834069.52      1600651.63      6834121.51
#Sta/Elev= 30
  4113.7 1742.84  4353.7 1736.46  4411.9 1736.71  4494.9 1732.81  4607.7 1729.69
  4655.4 1725.33  4695.5 1723.93  4857.6 1720.43    4962 1721.54  4967.5 1721.23
  4969.5 1708.84    4971 1707.84  5030.6 1708.84  5037.2 1708.99  5060.4 1721.37
  5219.9 1721.17  5390.9 1720.14  5477.3 1719.94  5536.3 1716.47  5569.2 1720.57
  5667.7 1718.61  6124.9 1723.84  6143.4 1724.04  6182.7 1729.45  6193.5  1729.6
  6263.7 1743.56  6303.9 1747.16  6393.9 1752.26  6461.7 1754.25  6831.3  1761.8
#Mann= 9 ,-1 , 0
  4113.7     .05       0  4494.9     .12       0  4969.5     .07       0
  5030.6     .12       0  5219.9     .05       0  5390.9     .12       0
  6124.9     .05       0  6303.9     .12       0  6461.7     .05       0
Bank Sta=4969.5,5030.6
XS Rating Curve= 0 ,0
Exp/Cntr=0.3,0.1

Type RM Length L Ch R = 1 ,17910   ,879,879,879
BEGIN DESCRIPTION:
Mapping XS 22398246
END DESCRIPTION:
XS GIS Cut Line= 4
      1597950.05       6833751.8      1598413.62      6834027.86
      1599627.16      6834293.48      1600679.29      6834350.78
#Sta/Elev= 30
    4090 1739.42    4171  1740.7  4383.2 1733.35    4582 1722.76  4681.7 1720.54
  4948.3 1719.69  4958.5 1718.88  4968.8 1715.04  4969.4 1709.93  4970.9 1708.93
  5030.6 1709.93  5031.5 1712.27  5050.7 1717.73  5070.3 1720.26  5341.5  1718.8
  5495.4 1719.12  5562.5 1716.41    5667 1718.87  5849.1 1720.86    5989 1719.26
    6088 1720.35    6187    1722  6320.3  1724.4  6400.4 1729.33  6460.5 1735.68
  6500.6 1746.88  6560.7 1752.68  6605.7 1753.55  6616.2  1753.9  6925.5 1759.81
#Mann= 12 ,-1 , 0
    4090     .05       0    4582     .12       0  4681.7     .05       0
  4969.4     .07       0  5030.6     .05       0  5341.5     .05       0
    5667     .12       0    5989     .05       0    6088     .12       0
    6187     .05       0  6605.7     .12       0  6616.2     .05       0
Bank Sta=4969.4,5030.6
XS Rating Curve= 0 ,0
Exp/Cntr=0.3,0.1

Type RM Length L Ch R = 1 ,17031   ,1081,1081,1081
BEGIN DESCRIPTION:
Mapping XS 42768128
END DESCRIPTION:
XS GIS Cut Line= 4
      1597564.63      6834085.13      1598455.29      6834605.98
      1599444.87      6835152.86      1599700.05        6835908.
#Sta/Elev= 30
  3356.6 1739.02  3774.1 1737.21  3805.5 1733.48  3891.5 1732.69  3971.6 1727.39
  4040.2 1726.93  4302.2 1717.02  4898.3 1718.48  4941.3 1718.89  4963.1 1717.08
  4969.4 1708.77  4970.9 1707.77  5030.7 1708.77  5038.7 1720.14  5102.3 1717.97
  5176.4 1717.77  5207.1 1715.03  5288.4 1717.86  5427.8 1716.54  5569.1 1719.03
  5663.5 1726.44  5726.4 1727.74  5767.2 1730.83  5789.3 1733.21  5815.4 1738.88
  5820.7  1737.8  5846.9 1746.74  5878.3 1750.15  5978.3 1753.13  6316.1 1756.48
#Mann= 5 ,-1 , 0
  3356.6     .05       0  4898.3     .12       0  4969.4     .07       0
  5030.7     .12       0  5102.3     .05       0
Bank Sta=4969.4,5030.7
XS Rating Curve= 0 ,0
Exp/Cntr=0.3,0.1

Type RM Length L Ch R = 1 ,15950   ,858,858,858
BEGIN DESCRIPTION:
Mapping XS e763e8b1
END DESCRIPTION:
XS GIS Cut Line= 4
      1597340.71      6834277.86      1597892.79      6834824.73
      1598950.08      6835632.02       1599585.5      6836569.54
#Sta/Elev= 30
  3950.6 1736.81  4295.4 1736.95  4396.1 1737.27  4505.3 1736.99  4660.8 1730.56
  4788.9 1728.98  4874.1 1725.01  4959.4 1719.52  4967.6 1717.31  4969.4 1708.02
  4970.9 1707.02  5030.7 1708.02  5059.1 1712.24  5067.4 1716.72  5089.3  1717.2
  5123.5 1714.37  5158.9  1717.1  5325.7 1717.25    5695 1715.45  5938.1 1720.66
  6015.1 1728.54  6037.9 1727.88  6051.6 1731.25  6057.9 1734.88  6065.2 1733.98
  6088.4 1743.32  6124.3 1747.67  6246.4 1751.94  6837.2 1755.27  7190.5 1754.94
#Mann= 7 ,-1 , 0
  3950.6     .05       0  4295.4     .12       0  4396.1     .05       0
  4969.4     .05       0  5030.7     .05       0  5089.3     .12       0
  5325.7     .05       0
Bank Sta=4969.4,5030.7
XS Rating Curve= 0 ,0
Exp/Cntr=0.3,0.1

Type RM Length L Ch R = 1 ,15092   ,463,463,463
BEGIN DESCRIPTION:
Mapping XS 8fef07ec
END DESCRIPTION:
XS GIS Cut Line= 4
      1597101.14      6834777.87       1597840.7      6835449.73
      1598663.62      6836402.86      1598799.03      6836642.44
#Sta/Elev= 30
  3574.8 1735.05  3747.5 1733.08  3782.7  1734.2  3818.4 1732.65  4094.1 1732.65
  4193.5 1729.77  4207.6 1730.68    4307 1725.86  4356.3 1726.11  4455.6 1720.95
  4561.7 1720.39  4783.5 1715.65  4853.4 1715.47  4958.4  1717.4  4966.1 1715.27
  4969.4 1709.23  4970.9 1708.23  5030.7 1709.23  5086.7 1714.65  5142.7 1714.69
  5234.9 1719.63  5263.4 1724.69  5298.5 1736.61  5334.7 1743.44  5363.2 1745.97
    5384 1744.94  5398.3 1747.39  5433.4 1749.39  5867.2 1752.32  6108.4 1750.79
#Mann= 5 ,-1 , 0
  3574.8     .05       0  4783.5      .1       0  4853.4     .12       0
  4969.4     .07       0  5030.7     .05       0
Bank Sta=4969.4,5030.7
XS Rating Curve= 0 ,0
Exp/Cntr=0.3,0.1

Type RM Length L Ch R = 1 ,14629   ,344,344,344
BEGIN DESCRIPTION:
Mapping XS f29a74ee
END DESCRIPTION:
XS GIS Cut Line= 4
      1596865.04      6835204.97      1597594.17      6835829.94
      1597986.54      6836312.58      1598299.06      6836680.67
#Sta/Elev= 30
  3780.2 1734.65  3902.7 1734.16  4267.8 1725.19  4372.4 1727.12  4522.5 1722.87
  4527.7 1722.71  4590.2  1721.9  4670.5 1715.83  4767.9 1713.93  4924.5 1716.12
  4950.9 1709.54  4969.2 1708.99  4970.7 1707.99  5030.8 1708.99  5031.6 1716.52
  5137.5 1721.72  5194.6 1735.61  5244.1 1741.48    5316 1742.18  5336.8 1745.99
  5351.2 1743.85    5372 1746.84  5379.8 1745.26  5386.3  1747.6  5394.1  1745.4
  5414.9 1747.98  5443.5 1745.54  5507.2 1749.21  5521.4 1746.87  5845.4 1749.82
#Mann= 9 ,-1 , 0
  3780.2     .05       0  4267.8     .12       0  4372.4     .05       0
  4522.5     .12       0  4527.7     .05       0  4670.5      .1       0
  4950.9     .05       0  4969.2     .05       0  5030.8     .05       0
Bank Sta=4969.2,5030.8
XS Rating Curve= 0 ,0
Exp/Cntr=0.3,0.1

Type RM Length L Ch R = 1 ,14285   ,284,284,284
BEGIN DESCRIPTION:
Mapping XS 96a4ea7a
END DESCRIPTION:
XS GIS Cut Line= 4
      1596135.82      6835329.93       1597153.2       6835909.8
      1597642.79      6836364.66      1597913.62        6836698.
#Sta/Elev= 30
  3384.2 1735.03  3402.2 1734.87  3631.7 1732.22    3661 1734.61  3911.2 1734.79
    3963 1732.75    4212 1734.91  4430.7 1729.18  4583.7 1718.14  4633.1 1721.93
  4654.1 1718.04  4703.9 1716.13  4866.6 1717.73  4913.4 1714.84  4930.1  1710.8
  4954.3 1709.12  4969.2 1709.08  4970.7 1708.08  5030.8 1709.08  5036.2 1718.16
  5064.5 1723.46  5176.8  1725.8  5247.2 1736.42  5348.1 1743.23  5376.8 1740.88
  5426.4 1743.33  5440.7 1741.24  5504.7 1744.44    5519 1742.77    5653 1745.53
#Mann= 10 ,-1 , 0
  3384.2      .1       0  3402.2     .05       0    3661    .075       0
    3963     .05       0  4913.4    .075       0  4954.3     .05       0
  4969.2     .03       0  5030.8     .05       0  5176.8    .075       0
  5247.2     .05       0
Bank Sta=4969.2,5030.8
XS Rating Curve= 0 ,0
Exp/Cntr=0.3,0.1

Type RM Length L Ch R = 1 ,14001   ,238,238,238
BEGIN DESCRIPTION:
Mapping XS ac820d99
END DESCRIPTION:
XS GIS Cut Line= 5
      1596045.55      6836236.19      1597010.84      6836316.05
      1597448.34      6836382.02      1597635.84      6836451.47
      1597906.67       6836722.3
#Sta/Elev= 30
  3797.4  1732.2  3917.3 1730.44  3987.5  1727.2  4077.8 1730.08  4268.5 1727.42
  4358.8 1724.44    4429 1719.67  4459.1 1712.49  4499.2 1709.45  4699.9 1709.35
  4780.3 1710.79  4809.1 1714.25  4814.1 1716.37  4861.2 1719.19  4911.8  1716.6
    4947 1709.37  4969.2 1709.05  4970.7 1708.05  5029.4 1708.05  5030.9 1709.05
  5033.1 1710.85  5079.8 1715.79  5093.8 1720.22  5103.9 1721.56  5143.6 1723.98
  5235.8 1726.46  5301.9 1731.53  5582.1 1742.37  5688.2  1744.6  5791.4 1744.89
#Mann= 3 ,-1 , 0
  3797.4     .05       0  4969.2     .03       0  5030.9     .05       0
Bank Sta=4969.2,5030.9
XS Rating Curve= 0 ,0
Exp/Cntr=0.3,0.1

Type RM Length L Ch R = 1 ,13763   ,712,712,712
BEGIN DESCRIPTION:
Mapping XS d7a37edd
END DESCRIPTION:
XS GIS Cut Line= 3
       1595944.9      6836559.11      1597476.12      6836524.39
      1597913.59      6836777.84
#Sta/Elev= 30
  3846.5 1735.25  4146.7  1734.7  4166.7 1738.18  4186.7 1734.47  4336.7 1732.31
  4406.7 1721.72  4456.8 1716.53  4536.8 1711.02  4586.8 1710.12  4596.8 1709.39
  4606.8  1706.3  4969.2  1706.3  4970.7  1705.3  5030.9  1706.3  5056.9 1712.42
  5066.9  1716.7  5116.9 1721.01  5156.9 1730.63    5237 1731.71    5297 1735.59
    5423 1734.97  5453.5  1739.7  5496.6 1741.37    5673 1744.24  5759.2 1743.77
  5769.1 1745.17  5774.9  1743.9  5790.7 1745.64  5862.2 1744.37  5883.7  1745.3
#Mann= 3 ,-1 , 0
  3846.5     .05       0  4969.2     .03       0  5030.9     .05       0
Bank Sta=4969.2,5030.9
XS Rating Curve= 0 ,0
Exp/Cntr=0.3,0.1

Type RM Length L Ch R = 1 ,13051   ,662,662,662
BEGIN DESCRIPTION:
Lytle Creek 13051.031
END DESCRIPTION:
XS GIS Cut Line= 3
        1596105.        6836838.      1596613.14      6837031.94
      1597405.02        6837038.
#Sta/Elev= 30
  4456.1 1738.37  4488.2 1736.98  4501.2 1735.35  4586.1 1732.96  4659.5 1728.27
  4702.3 1723.19  4780.6  1716.1  4787.9 1712.64  4810.7 1710.77    4820 1707.82
    4830  1706.3  4969.2  1706.3  4970.7  1705.3  5029.4  1705.3  5030.9  1706.3
  5181.9  1706.3  5191.9 1709.75  5221.9  1715.7  5281.9 1717.94  5311.9 1716.05
  5331.9 1711.24  5361.9 1711.24  5401.9 1724.52  5411.9 1725.84  5461.9 1726.53
  5491.9 1730.09  5521.9 1731.43  5621.9 1732.09  5691.9 1734.82  5791.9  1736.7
#Mann= 3 ,-1 , 0
  4456.1     .05       0  4969.2     .03       0  5030.9     .05       0
Bank Sta=4969.2,5030.9
XS Rating Curve= 0 ,0
Exp/Cntr=0.3,0.1

Type RM Length L Ch R = 1 ,12389   ,492,492,492
BEGIN DESCRIPTION:
Mapping XS bc94589d
END DESCRIPTION:
XS GIS Cut Line= 3
      1595687.96       6837746.6       1597191.4        6837573.
      1598274.72      6837479.25
#Sta/Elev= 30
  4127.5 1730.44  4215.1 1729.02  4509.8 1728.26  4593.7 1725.59  4688.2 1719.97
  4738.6  1718.3  4766.4 1716.01  4778.8 1712.09    4809 1710.78  4819.1 1707.24
  4829.2  1706.3  4969.2  1706.3  4970.7  1705.3  5029.4  1705.3  5030.9  1706.3
  5205.8  1706.3  5211.7 1709.05  5231.8 1710.93  5241.9 1716.42  5332.5 1730.61
    5564 1732.74  5845.3 1738.96  5989.8 1739.17    6036 1741.28    6307 1742.88
  6457.7 1745.23  6507.8 1743.65  6618.2 1747.84  6698.5 1746.54  6728.3 1747.33
#Mann= 3 ,-1 , 0
  4127.5     .05       0  4969.2     .03       0  5030.9     .05       0
Bank Sta=4969.2,5030.9
XS Rating Curve= 0 ,0
Exp/Cntr=0.3,0.1

Type RM Length L Ch R = 1 ,11897   ,620,620,620
BEGIN DESCRIPTION:
Mapping XS fcdb02d6
END DESCRIPTION:
XS GIS Cut Line= 3
      1595739.98      6838191.05      1597344.17      6838045.22
      1598374.47      6837812.79
#Sta/Elev= 30
  4081.9 1728.02  4147.2 1726.82  4171.6 1728.63  4187.4 1726.71  4237.6 1726.16
  4287.8 1729.05  4327.9  1726.4  4629.2 1728.69  4723.8 1719.74  4739.6 1714.23
  4769.7 1711.01  4789.8  1706.3  4969.2  1706.3  4970.7  1705.3  5030.9  1706.3
  5160.6 1706.53  5171.4 1710.08  5211.6 1713.26  5231.6 1723.97  5241.7 1720.62
  5261.8 1721.97  5342.1 1734.71  5939.6 1741.24  6011.3 1739.75  6052.4 1741.68
  6359.9 1741.74  6452.2 1745.09  6519.8 1742.52  6554.7 1746.13  6748.9 1747.88
#Mann= 3 ,-1 , 0
  4081.9     .05       0  4969.2     .03       0  5030.9     .05       0
Bank Sta=4969.2,5030.9
XS Rating Curve= 0 ,0
Exp/Cntr=0.3,0.1

Type RM Length L Ch R = 1 ,11277   ,789,789,789
BEGIN DESCRIPTION:
Mapping XS 984a383e
END DESCRIPTION:
XS GIS Cut Line= 3
       1595736.5      6838704.94       1597528.2      6838691.05
      1598635.88      6838225.76
#Sta/Elev= 30
  3981.8 1725.55  4005.7 1725.64  4340.3 1727.58  4420.3 1726.63  4480.3 1724.66
  4560.3 1717.82  4610.3  1706.3  4969.2  1706.3  4970.7  1705.3  5029.4  1705.3
  5030.9  1706.3  5350.3  1706.3  5370.3 1710.76  5380.3 1716.11  5410.3 1718.61
  5470.3 1727.68  5570.4 1733.79  5835.2 1736.36    5867 1735.37  5996.7 1736.18
  6214.8 1739.29  6279.7 1737.15  6314.3 1738.68  6361.8 1736.56  6367.2 1737.54
  6449.9 1736.57  6462.7 1736.73  6544.4 1735.98    6768 1744.13    6975 1746.25
#Mann= 6 ,-1 , 0
  3981.8    .075       0  4005.7     .05       0  4969.2     .03       0
  5030.9     .05       0  6449.9    .075       0  6462.7     .05       0
Bank Sta=4969.2,5030.9
XS Rating Curve= 0 ,0
Exp/Cntr=0.3,0.1

Type RM Length L Ch R = 1 ,10488   ,771,771,771
BEGIN DESCRIPTION:
Mapping XS 10ce9f81
END DESCRIPTION:
XS GIS Cut Line= 6
      1595596.12      6839023.72      1595999.77      6839427.38
      1597041.44      6839470.78      1597280.16      6839188.67
      1597579.63      6839002.03      1598669.02      6838385.73
#Sta/Elev= 30
  3773.3  1722.8  4079.6 1725.59  4344.2 1724.19  4409.4 1722.04  4459.5 1716.67
  4529.5 1715.28  4569.6 1711.47  4589.6  1706.3  4969.2  1706.3  4970.7  1705.3
  5030.9  1706.3  5380.3  1706.3  5419.3  1711.1  5433.6 1716.66    5483 1727.07
    5505 1728.55  5840.6 1727.26  5861.8 1729.14  5919.7 1728.04  6599.1 1738.24
  6674.2 1736.75  6724.4 1738.94  6751.4 1739.16  6856.7  1738.6  6895.1 1740.72
  6954.1 1740.19  6988.5 1735.64  7036.3 1737.77  7084.1 1741.36  7360.8 1745.24
#Mann= 7 ,-1 , 0
  3773.3     .05       0  4969.2     .03       0  5030.9     .05       0
  6724.4    .075       0  6751.4     .05       0  6856.7    .075       0
  7036.3     .05       0
Bank Sta=4969.2,5030.9
XS Rating Curve= 0 ,0
Exp/Cntr=0.3,0.1

Type RM Length L Ch R = 1 ,9717    ,316,316,316
BEGIN DESCRIPTION:
Mapping XS c2292043
END DESCRIPTION:
XS GIS Cut Line= 5
      1595296.64      6840069.74      1595982.41      6840217.31
      1597488.49      6840234.67      1597853.07      6840416.96
      1598801.78      6840347.65
#Sta/Elev= 30
  3625.9 1725.32  3739.2 1721.38  4012.9 1718.77  4094.7 1719.93  4212.1 1717.75
  4227.7  1714.3    4238 1713.91  4299.3 1713.98    4410 1710.41    4430  1706.3
  4968.9  1706.3  4970.4  1705.3  5029.6  1705.3  5031.1  1706.3    5680  1706.3
  5686.8 1709.91  5691.8 1709.35    5710 1712.95    5740 1722.62  5780.1 1725.21
  5810.1 1725.65  6011.4 1727.18  6333.3  1727.1  6353.4 1728.38  6553.9  1729.4
  6914.9  1730.1  6924.9 1729.29    6965 1730.38  7165.5 1729.99  7192.4 1730.94
#Mann= 3 ,-1 , 0
  3625.9     .05       0  4968.9     .03       0  5031.1     .05       0
Bank Sta=4968.9,5031.1
XS Rating Curve= 0 ,0
Exp/Cntr=0.3,0.1

Type RM Length L Ch R = 1 ,9401    ,427,427,427
BEGIN DESCRIPTION:
Mapping XS 3c507853
END DESCRIPTION:
XS GIS Cut Line= 4
      1595283.99      6840340.62      1596390.72      6840518.56
       1597853.4      6840644.43      1598799.54      6840444.79
#Sta/Elev= 30
  3613.8 1723.89  3758.2 1722.34  3857.9 1719.35  3938.8 1720.82  4030.1 1720.09
  4040.2  1718.8  4080.7 1720.11  4273.2 1717.65  4283.3 1716.43  4303.6  1706.3
  4968.9  1706.3  4970.4  1705.3  5029.6  1705.3  5031.1  1706.3  5702.6  1706.3
  5712.6 1706.83  5718.6 1710.33  5732.7 1711.42  5752.8 1720.04  5762.8 1721.48
  6003.7 1727.14  6259.4 1728.37  6541.7 1726.39  6623.5 1727.15  6642.2 1726.26
  6746.9 1727.72    6879 1727.67  6919.9 1729.16  7129.7 1728.94  7169.8 1729.94
#Mann= 3 ,-1 , 0
  3613.8     .05       0  4968.9     .03       0  5031.1     .05       0
Bank Sta=4968.9,5031.1
XS Rating Curve= 0 ,0
Exp/Cntr=0.3,0.1

Type RM Length L Ch R = 1 ,8974    ,639,639,639
BEGIN DESCRIPTION:
Mapping XS f694fd06
END DESCRIPTION:
XS GIS Cut Line= 4
      1595296.92      6840462.13      1595895.93      6840540.26
      1596859.47      6841117.52       1598070.2       6842037.5
#Sta/Elev= 30
  3627.8 1725.32  3676.3 1724.67  3706.5 1722.81  3785.7 1722.95  3817.5 1720.91
  3908.2 1720.61  4022.6 1718.33    4120 1719.43  4242.7 1717.78  4258.3 1716.83
  4273.9  1706.3  4968.8  1706.3  4970.3  1705.3  5029.7  1705.3  5031.2  1706.3
    5595  1706.3  5601.3 1709.59  5609.5 1709.29  5624.1 1711.16  5630.3 1713.92
  5638.4 1714.94  5644.9 1717.47  5659.4 1720.51  5694.8 1722.62  6008.8 1726.08
  6087.8 1725.64  6229.3 1727.42  6434.2 1727.72  6465.7 1728.06  6875.7 1731.49
#Mann= 5 ,-1 , 0
  3627.8     .05       0  4968.8     .03       0  5031.2     .05       0
  6434.2    .075       0  6465.7     .05       0
Bank Sta=4968.8,5031.2
XS Rating Curve= 0 ,0
Exp/Cntr=0.3,0.1

Type RM Length L Ch R = 1 ,8335    ,755,755,755
BEGIN DESCRIPTION:
Mapping XS 9461dd3d
END DESCRIPTION:
XS GIS Cut Line= 3
      1595288.33      6840761.64      1597232.74      6842215.61
      1597775.26      6842515.08
#Sta/Elev= 30
  3897.8 1726.51  4006.3 1724.63  4029.2 1722.62  4364.8 1721.44  4456.5 1719.38
  4535.7 1720.55  4592.9 1719.66  4621.1 1712.18  4664.9 1708.43  4671.1  1706.3
  4968.8  1706.3  4970.3  1705.3  5029.7  1705.3  5031.2  1706.3  5406.9  1706.3
  5415.2 1712.09  5429.5  1714.6    5436 1717.85  5442.3 1718.81  5679.2 1725.02
    5807 1723.98  5850.8 1725.23  5900.8 1724.01  6100.9  1726.4  6142.6 1725.23
  6307.2 1728.21  6533.9 1728.02  6843.5 1733.07  6892.3 1732.98  6945.4 1733.16
#Mann= 5 ,-1 , 0
  3897.8     .05       0  4968.8     .03       0  5031.2     .05       0
  6843.5    .075       0  6892.3     .05       0
Bank Sta=4968.8,5031.2
XS Rating Curve= 0 ,0
Exp/Cntr=0.3,0.1

Type RM Length L Ch R = 1 ,7580    ,513,513,513
BEGIN DESCRIPTION:
Mapping XS 5a191e74
END DESCRIPTION:
XS GIS Cut Line= 4
      1594906.37      6841169.63      1595301.31      6841712.14
      1596325.62      6842432.62      1597158.98      6842818.92
#Sta/Elev= 30
  3833.1 1722.45  3843.8 1722.63  4160.5 1720.77  4302.7    1717  4403.1 1719.41
  4482.7 1718.57  4518.9 1717.25  4533.1 1714.31  4539.8 1710.79  4575.5  1706.3
  4968.8  1706.3  4970.3  1705.3  5031.2  1706.3  5450.2  1706.3    5465 1711.63
  5494.6 1713.87  5500.7 1716.91  5515.5 1717.86  5559.9 1717.24  5566.1 1715.01
  5601.8  1712.5  5616.6 1715.78  5622.7 1714.27  5652.3 1716.97  5782.2 1717.09
  5805.1 1721.33  6097.5 1720.22  6228.6 1723.93  6377.1 1723.07    6675 1727.85
#Mann= 4 ,-1 , 0
  3833.1    .075       0  3843.8     .05       0  4968.8     .03       0
  5031.2     .05       0
Bank Sta=4968.8,5031.2
XS Rating Curve= 0 ,0
Exp/Cntr=0.3,0.1

Type RM Length L Ch R = 1 ,7067    ,570,570,570
BEGIN DESCRIPTION:
Mapping XS 61d46f32
END DESCRIPTION:
XS GIS Cut Line= 4
      1594841.24      6841864.04      1595166.77      6842159.19
      1596169.37       6843001.2      1596512.22      6843274.61
#Sta/Elev= 30
  4115.5 1721.34  4152.6 1721.14  4166.7 1720.22  4177.4 1718.03  4191.6 1717.46
  4302.9 1716.03    4404 1715.02  4427.4 1713.03  4432.2 1714.03  4439.6 1711.78
  4446.4 1712.91  4453.8  1711.2  4474.8 1710.29  4482.2 1708.27    4489 1709.13
  4496.4  1706.3  4968.8  1706.3  4970.3  1705.3  5031.2  1706.3  5461.4  1706.3
  5475.7 1709.72  5525.2 1712.44    5546 1717.24  5695.6 1720.01  5930.1 1717.91
  5958.9 1718.28  5979.7  1720.5  6037.4 1718.66    6079 1720.04  6302.7 1719.98
#Mann= 7 ,-1 , 0
  4115.5     .05       0  4152.6     .12       0  4166.7     .05       0
  4302.9     .12       0  4427.4     .05       0  4968.8     .03       0
  5031.2     .05       0
Bank Sta=4968.8,5031.2
XS Rating Curve= 0 ,0
Exp/Cntr=0.3,0.1

Type RM Length L Ch R = 1 ,6497    ,76,76,76
BEGIN DESCRIPTION:
Mapping XS e246b9a7
END DESCRIPTION:
XS GIS Cut Line= 6
      1594839.08        6841914.      1594888.99      6842608.41
      1595014.86      6842749.47      1595490.12      6843046.77
      1595900.27      6843246.43      1596451.84      6843438.93
#Sta/Elev= 30
  3708.7 1721.88  3742.8 1721.95  3762.9 1719.33  3781.3 1719.03  4104.3 1717.46
  4164.4 1714.39  4204.4 1709.12  4212.1  1706.3  4815.9  1706.3  4875.4  1706.3
  4968.8  1706.3  4970.3  1705.3  5029.7  1705.3  5031.2  1706.3  5452.8  1706.3
  5459.2 1706.96  5469.3 1709.68  5497.1 1711.33  5519.2 1714.23  5535.7  1719.2
  5541.3 1719.59  5602.1 1718.15    5632 1719.24  5657.8 1718.01  5669.6 1716.52
  5711.9 1716.46  5844.2 1717.29  5994.2 1719.39  6180.5 1719.46  6195.8 1720.45
#Mann= 6 ,-1 , 0
  3708.7     .12       0  3781.3     .05       0  4815.9     .12       0
  4875.4     .05       0  4968.8     .03       0  5031.2     .05       0
Bank Sta=4968.8,5031.2
XS Rating Curve= 0 ,0
Exp/Cntr=0.3,0.1

Type RM Length L Ch R = 1 ,6421    ,102,102,102
BEGIN DESCRIPTION:
Mapping XS 61c250d7
END DESCRIPTION:
XS GIS Cut Line= 6
      1594817.37      6841937.79      1594841.24      6842202.59
      1594832.56      6842723.42      1594871.63      6842779.85
      1595963.21      6843370.12      1596457.98      6843478.63
#Sta/Elev= 30
  3600.4 1720.88  3648.4  1718.7  4771.5 1722.25  4826.6 1716.72    4859  1721.5
  4884.3 1722.55  4964.9 1722.62  4968.8  1706.3  4970.3  1705.3  5031.2  1706.3
  5032.4 1722.59  5039.8 1722.87  5153.9 1722.72  5197.5 1707.48  5239.4 1714.51
  5245.1  1706.5  5274.7 1712.22  5282.7 1707.13  5297.6    1713  5304.4  1706.3
  5320.4 1713.77  5326.1 1707.83    5342  1712.3  5369.4 1708.42  5377.9 1713.45
    5481 1710.06  5503.6 1712.48  5520.6 1721.21  5808.6 1716.72  6207.1 1720.65
#Mann= 7 ,-1 , 0
  3600.4     .12       0  3648.4     .05       0  4771.5     .12       0
    4859     .05       0  4884.3     .12       0  4968.8     .05       0
  5031.2     .05       0
Bank Sta=4968.8,5031.2
XS Rating Curve= 0 ,0
Exp/Cntr=0.3,0.1

Type RM Length L Ch R = 1 ,6319    ,340,340,340
BEGIN DESCRIPTION:
Mapping XS b8d173da
END DESCRIPTION:
XS GIS Cut Line= 5
      1593977.12      6842469.97      1594772.23      6842924.81
      1595091.68      6843018.56      1595796.54      6843390.09
      1596413.92      6843643.28
#Sta/Elev= 30
  3508.6  1713.8  3792.5 1714.61  4099.1 1712.51  4222.9 1715.69  4448.3 1715.62
  4479.6 1714.89    4559 1706.84  4592.4  1708.2  4677.8 1706.61  4729.7  1704.5
  4750.6 1701.39  4816.8 1699.67    4874 1699.61  4937.6 1698.45  4953.5 1694.94
  4968.8 1694.39  4970.3 1693.39  5031.2 1694.39  5032.6  1696.8  5037.4 1697.49
    5123 1699.67  5174.2 1707.49  5190.6 1703.88  5322.7 1706.92  5476.9 1706.65
    5499 1716.08  5515.3 1716.92  5821.5 1716.15  6157.9 1718.97  6221.6    1721
#Mann= 7 ,-1 , 0
  3508.6     .05       0  4677.8     .12       0  4816.8     .05       0
    4874     .12       0  4968.8     .07       0  5031.2     .12       0
  5037.4     .05       0
Bank Sta=4968.8,5031.2
XS Rating Curve= 0 ,0
Exp/Cntr=0.3,0.1

Type RM Length L Ch R = 1 ,5979    ,517,517,517
BEGIN DESCRIPTION:
Mapping XS 37e76429
END DESCRIPTION:
XS GIS Cut Line= 4
      1594068.66      6842658.31       1594706.7      6843088.01
      1595579.09      6843708.67      1596368.99      6843821.51
#Sta/Elev= 30
  3657.3  1713.9  3677.7  1713.8  3917.4 1713.92  3956.2 1712.91  4014.6 1714.32
  4166.1 1711.42  4181.1 1713.91    4397 1713.41  4518.9 1711.74  4628.2 1706.27
  4697.2  1704.8    4719 1699.81  4898.9 1698.55  4951.5 1694.85  4964.1  1694.6
  4968.8 1692.26  4970.3 1691.26  5031.3 1692.26  5035.4 1695.57  5099.9 1697.23
  5121.5 1702.19  5127.6 1705.54  5200.1 1708.16  5234.6 1710.78  5329.3 1713.27
  5492.3  1715.4  5715.3 1714.51    5786 1717.78  5907.2 1716.89  6295.1 1721.25
#Mann= 9 ,-1 , 0
  3657.3     .05       0  3677.7    .075       0  3917.4     .05       0
  4628.2     .12       0  4951.5     .05       0  4968.8     .03       0
  5031.3     .05       0  5099.9     .12       0  5200.1     .05       0
Bank Sta=4968.8,5031.3
XS Rating Curve= 0 ,0
Exp/Cntr=0.3,0.1

Type RM Length L Ch R = 1 ,5462    ,411,411,411
BEGIN DESCRIPTION:
Mapping XS 6eee6da3
END DESCRIPTION:
XS GIS Cut Line= 4
      1593532.65      6843483.84      1594209.73       6843664.4
      1595550.01      6843931.76      1596361.28      6843928.29
#Sta/Elev= 30
  3648.6 1714.47    3858 1715.43  4306.7 1709.55    4494 1709.94  4528.1 1706.38
  4609.6 1705.52    4677 1700.51  4703.3  1697.2  4754.3 1695.44  4864.6 1697.24
  4907.5 1691.56  4935.9 1695.78  4953.4  1691.8  4968.8  1691.3  4970.3  1690.3
  5031.3  1691.3  5037.9 1696.52  5060.6 1697.71    5221 1701.22  5252.1 1701.51
  5264.8 1703.76  5374.4 1702.29  5486.6 1704.68  5617.1 1710.91    5716 1713.27
  5890.2 1712.08    6001 1716.61  6213.4 1718.39  6438.4 1721.06  6527.3 1721.66
#Mann= 8 ,-1 , 0
  3648.6     .05       0    4677     .12       0  4968.8     .07       0
  5031.3     .12       0    5221     .05       0  5890.2    .075       0
  6213.4     .05       0  6438.4    .075       0
Bank Sta=4968.8,5031.3
XS Rating Curve= 0 ,0
Exp/Cntr=0.3,0.1

Type RM Length L Ch R = 1 ,5051    ,635,635,635
BEGIN DESCRIPTION:
Mapping XS a91f2043
END DESCRIPTION:
XS GIS Cut Line= 4
      1593303.26      6843925.41      1594136.57      6843967.07
      1594891.78      6844071.24      1595646.94      6844138.94
#Sta/Elev= 30
  3776.8 1711.84  3888.7 1712.08  3926.3 1713.61  4009.1 1712.96  4126.5 1711.38
  4144.5 1712.16  4339.2 1711.61  4579.5 1707.43  4607.9 1703.04  4654.8 1700.42
  4791.3 1698.61  4875.6  1695.5  4902.3 1697.01  4922.5 1695.06  4942.5  1691.5
  4968.7 1691.25  4970.2 1690.25  5029.8 1690.25  5031.3 1691.25  5043.6 1691.28
  5063.8 1695.94  5073.9  1696.7    5185 1698.69  5225.3  1703.4  5255.6 1704.67
  5306.1 1704.07  5537.4  1710.1  5828.5 1710.68  5898.8 1709.94  6131.7 1712.66
#Mann= 5 ,-1 , 0
  3776.8     .05       0  4009.1    .075       0  4144.5     .05       0
  4968.7     .05       0  5031.3     .05       0
Bank Sta=4968.7,5031.3
XS Rating Curve= 0 ,0
Exp/Cntr=0.3,0.1

Type RM Length L Ch R = 1 ,4416    ,456,456,456
BEGIN DESCRIPTION:
Mapping XS 28d35157
END DESCRIPTION:
XS GIS Cut Line= 3
      1593256.33      6844039.97      1594725.11      6844784.78
      1594865.73      6844821.24
#Sta/Elev= 30
    4033  1711.3  4088.6 1710.47  4210.9 1710.91    4267 1712.36    4634 1705.37
  4737.9 1705.21    4879 1700.63  4923.5 1696.42  4945.8 1695.06    4968 1695.08
  4968.7 1691.17  4970.2 1690.17  5029.8 1690.17  5031.3 1691.17  5057.1 1691.17
    5063 1694.57  5073.8  1695.3  5168.5 1696.44  5257.5 1696.33  5279.8 1697.78
  5296.5 1696.63  5318.7 1697.04  5354.6  1699.8  5407.8 1701.49  5541.4 1704.87
  5569.3  1704.8  5585.9 1706.64  5623.7 1706.18  5668.5 1707.05  5825.1 1711.75
#Mann= 3 ,-1 , 0
    4033     .05       0  4968.7     .05       0  5031.3     .05       0
Bank Sta=4968.7,5031.3
XS Rating Curve= 0 ,0
Exp/Cntr=0.3,0.1

Type RM Length L Ch R = 1 ,3960    ,483,483,483
BEGIN DESCRIPTION:
Mapping XS e9e981e6
END DESCRIPTION:
XS GIS Cut Line= 3
      1592652.22      6844362.91      1594745.95      6845196.24
       1595100.1      6845258.74
#Sta/Elev= 30
    3589 1700.24  3623.5 1700.41  3671.5 1699.44  3720.1 1700.95  3778.7 1700.83
  3907.7 1699.98  4049.2 1698.72  4162.5 1700.66  4186.7  1697.9    4211  1699.4
    4476 1697.22    4559 1696.36  4621.7 1697.55  4738.9 1698.39  4809.9 1698.96
  4872.8 1696.29  4958.9 1695.82  4966.3 1695.41  4968.7 1691.11  4970.2 1690.11
  5029.8 1690.11  5031.3 1691.11  5103.9 1691.44  5152.5 1694.61  5540.9 1699.89
  5667.7 1702.75    5673 1704.29  5756.7 1704.35  5780.9 1706.37  6202.1 1708.57
#Mann= 9 ,-1 , 0
    3589     .05       0  3623.5     .12       0  3778.7    .075       0
  3907.7     .12       0    4476     .05       0  4621.7     .12       0
  4738.9     .05       0  4968.7     .05       0  5031.3     .05       0
Bank Sta=4968.7,5031.3
XS Rating Curve= 0 ,0
Exp/Cntr=0.3,0.1

Type RM Length L Ch R = 1 ,3477    ,455,455,455
BEGIN DESCRIPTION:
Mapping XS 03b72a6c
END DESCRIPTION:
XS GIS Cut Line= 3
      1592490.76      6844816.04      1594495.95      6845581.66
      1594839.71      6845597.28
#Sta/Elev= 30
  3643.5 1699.63  3688.3 1697.06  3748.4 1697.34  3787.2 1696.17  3989.8 1696.75
  4367.2 1695.98  4397.3 1697.62    4422 1694.52    4537 1697.42  4547.2 1696.66
  4739.9 1696.51    4772 1695.02  4865.7 1697.53  4925.9  1694.7  4950.6 1695.09
  4955.9 1694.57  4964.6 1691.05  4968.7 1691.05  4970.2 1690.05  5029.9 1690.05
  5031.4 1691.05  5060.2 1691.05  5082.4 1694.36  5095.6  1694.9  5210.8 1697.49
    5405 1699.76    5679 1700.14    5829 1705.54  5949.1 1708.31    6134 1709.22
#Mann= 5 ,-1 , 0
  3643.5     .05       0  3989.8     .12       0  4367.2     .05       0
  4968.7     .03       0  5031.4     .05       0
Bank Sta=4968.7,5031.4
XS Rating Curve= 0 ,0
Exp/Cntr=0.3,0.1

Type RM Length L Ch R = 1 ,3022    ,325,325,325
BEGIN DESCRIPTION:
Mapping XS 52a88089
END DESCRIPTION:
XS GIS Cut Line= 4
      1592465.97       6844863.9      1592481.97      6845313.37
      1593938.66      6845816.03      1594691.95      6845826.42
#Sta/Elev= 30
  3451.7 1699.28    3766 1696.42  3876.1 1696.25  3905.7 1698.13  3925.8 1697.92
    3931 1696.46  4081.7 1695.07  4144.1 1696.33  4211.8 1695.04  4263.6  1696.1
  4581.7 1695.32    4638 1695.74  4655.7  1697.5  4669.2  1697.3  4676.9 1694.16
  4695.1 1695.79  4867.3 1695.61  4920.2 1694.63  4968.7 1690.98  4970.2 1689.98
  5031.4 1690.98  5068.5 1691.66  5078.9 1695.01  5110.6 1696.05  5157.7 1695.09
  5316.7 1696.51  5535.3 1698.44  6036.2 1704.62  6177.5  1706.1  6195.8 1706.03
#Mann= 8 ,-1 , 0
  3451.7     .05       0  4968.7     .07       0  5031.4     .05       0
  5068.5     .05       0  5316.7    .075       0  5535.3     .05       0
  6036.2    .075       0  6177.5      .1       0
Bank Sta=4968.7,5031.4
XS Rating Curve= 0 ,0
Exp/Cntr=0.3,0.1

Type RM Length L Ch R = 1 ,2697    ,236,236,236
BEGIN DESCRIPTION:
Mapping XS 53d90626
END DESCRIPTION:
XS GIS Cut Line= 5
      1592450.35      6844918.58      1592342.84      6845705.72
      1593032.41      6845862.91      1593865.74      6846071.24
      1594615.74      6846071.24
#Sta/Elev= 30
  3131.5 1698.42  4174.3 1694.45  4246.1 1695.59  4363.9 1693.69  4430.7 1694.82
  4769.9 1694.93  4780.2 1693.86  4790.5 1694.46  4797.1 1699.32  4802.2 1699.62
  4811.1  1699.5  4831.7 1693.68  4862.7 1695.26  4890.2 1694.64  4945.1 1694.78
  4955.4 1691.99  4968.7 1690.94  4970.2 1689.94  5029.9 1689.94  5031.4 1690.94
  5044.4 1690.94  5068.8 1695.32  5092.8 1696.93    5110 1694.84  5151.3 1694.59
  5333.1 1695.72  5410.1 1696.49  5811.5 1699.64    5993 1703.07  6242.2 1706.82
#Mann= 9 ,-1 , 0
  3131.5     .05       0  4890.2     .12       0  4968.7     .05       0
  5031.4     .12       0  5044.4     .12       0  5092.8     .05       0
  5333.1    .075       0  5410.1     .05       0    5993    .075       0
Bank Sta=4968.7,5031.4
XS Rating Curve= 0 ,0
Exp/Cntr=0.3,0.1

Type RM Length L Ch R = 1 ,2461    ,213,213,213
BEGIN DESCRIPTION:
Mapping XS e7afadb7
END DESCRIPTION:
XS GIS Cut Line= 6
       1592364.4       6845259.8      1592301.91      6845744.14
      1592341.48       6845873.1       1592839.7      6846076.45
      1593657.41      6846237.91      1594431.75      6846175.54
#Sta/Elev= 30
  3315.5 1697.19  3849.7 1696.45  4039.3 1695.21  4068.8 1694.66  4074.2 1693.49
  4127.6 1694.66    4353 1692.68  4765.7 1695.94  4798.2 1695.81  4828.8 1693.67
    4839 1695.65  4868.3 1693.82  4918.7 1694.38    4941 1690.91  4968.7 1690.91
  4970.2 1689.91  5029.9 1689.91  5031.4 1690.91  5042.9 1690.91  5073.4 1694.17
  5093.8 1698.45  5110.8 1697.11  5129.8 1694.02  5267.1 1693.81  5428.3 1697.13
  5508.6  1696.3  5669.1 1698.78  5819.6 1699.09  6018.7 1703.42  6087.2 1704.62
#Mann= 6 ,-1 , 0
  3315.5     .05       0  4918.7     .12       0  4968.7     .07       0
  5031.4     .12       0  5110.8     .05       0  6018.7    .075       0
Bank Sta=4968.7,5031.4
XS Rating Curve= 0 ,0
Exp/Cntr=0.3,0.1
