--- Lytle Creek.prj (project) ---

Proj Title=Lytle Creek Base Level Engineering
Current Plan=p02
Default Exp/Contr=0.3,0.1
English Units
Geom File=g01
Geom File=g02
Flow File=f01
Plan File=p01
Plan File=p02
Y Axis Title=Elevation
X Axis Title(PF)=Main Channel Distance
X Axis Title(XS)=Station
BEGIN DESCRIPTION:
Lytle Creek
END DESCRIPTION:
DSS Export Rating Curves= 0
DSS Export Rating Curve Sorted= 0
DSS Export Volume Flow Curves= 0
DXF OffsetX= 0
DXF OffsetY= 0
DXF ScaleX= 1
DXF ScaleY= 10

--- Lytle Creek.p02 (plan) ---

Plan Title=ohrlord
Program Version=4.10
Short Identifier=ohlord
Geom File=g02
Flow File=f01
Subcritical Flow
K Sum by GR= 0
Std Step Tol= 0.01
Critical Tol= 0.01
Num of Std Step Trials= 20
Max Error Tol= 0.3
Flow Tol Ratio= 0.001
Split Flow NTrial= 30
Split Flow Tol= 0.02
Split Flow Ratio= 0.02
Log Output Level= 0
Friction Slope Method= 1
Unsteady Friction Slope Method= 2
Unsteady Bridges Friction Slope Method= 1
Parabolic Critical Depth
Global Vel Dist= 1 , 1 , 1
Global Log Level= 0
CheckData=True
Encroach Param=-1 ,0,0, 0
BEGIN DESCRIPTION:
Multiple Run
END DESCRIPTION:
Computation Interval=1HOUR
Output Interval=1HOUR
Run HTab= 0
Run UNet= 0
Run PostProcess= 0
Run WQNet= 0
UNET Theta= 1
UNET Theta Warmup= 1
UNET ZTol= 0.02
UNET ZSATol= 0.05
UNET MxIter= 20
UNET MaxInSteps= 0
UNET DtIC= 0
UNET DtMin= 0
UNET MaxCRTS= 20
UNET WFStab= 2
UNET SFStab= 1
UNET WFX= 1
UNET SFX= 1
UNET DSS MLevel= 4
UNET DZMax Abort= 100
UNET Convert EG Bridges= 0
UNET Use Existing IB Tables=-1
UNET Froude Reduction=False
UNET Froude Limit= 1
UNET Froude Power= 10
UNET Time Slicing=0,0, 5
UNET Junction Losses=0
Instantaneous Interval=1HOUR
Write IC File= 0
Write IC File at Sim End=0
Echo Input=False
Echo Parameters=False
Echo Output=False
Write Detailed= 0
WQ AD Non Conservative
WQ ULTIMATE=-1
WQ Max Comp Step=1HOUR
WQ Output Interval=15MIN
WQ Output Selected Increments= 0
WQ Output face flow=0
WQ Output face velocity=0
WQ Output face area=0
WQ Output face dispersion=0
WQ Output cell volume=0
WQ Output cell surface area=0
WQ Output cell continuity=0
WQ Output cumulative cell continuity=0
WQ Output face conc=0
WQ Output face dconc_dx=0
WQ Output face courant=0
WQ Output face peclet=0
WQ Output face adv mass=0
WQ Output face disp mass=0
WQ Output cell mass=0
WQ Output cell source sink temp=0
WQ Output cell source sink nsm=0
WQ Output MaxMinRange=-1
WQ Daily Max Min Mean=-1
WQ Daily Range=0
WQ Daily Time=0
WQ Create Restart=0
WQ Fixed Restart=0
WQ System Summary=0
WQ Use Fixed Temperature=0
Sorting and Armoring Iterations= 10
XS Update Threshold= 0.02
Hydraulics Update Threshold= 0.02
Energy Slope Method= 1
Volume Change Method= 0
XS Weighting Method= 0
Number of US Weighted Cross Sections= 1
Number of DS Weighted Cross Sections= 1
Upstream XS Weight=0.25
Main XS Weight=0.5
Downstream XS Weight=0.25
Number of DS XS's Weighted with US Boundary= 1
Upstream Boundary Weight= 1
Weight of XSs Associated with US Boundary= 0
Number of US XS's Weighted with DS Boundary= 1
Downstream Boundary Weight= 0.5
Weight of XSs Associated with DS Boundary= 0.5
Sediment Output Level= 4
Mass or Volume Output= 0
Output Increment Type= 1
Profile and TS Output Increment= 10
XS Output Flag= 0
XS Output Increment= 10
Disregard all LS=0
Disregard all Conn=0
Disregard all Breaches=0
Disregard all Pumps=0

--- Lytle Creek.f01 (steady flow) ---

Flow Title=Multiple
Program Version=4.10
Number of Profiles= 7
Profile Names=10-year,25-year,50-year,1pct_min,100-year,1pct_plu,500-year
River Rch & RM=Lytle Creek,Reach-1         ,97944
     293     415     518     323     644    1286    1008
River Rch & RM=Lytle Creek,Reach-1         ,97699
     386     554     698     438     874    1744    1390
River Rch & RM=Lytle Creek,Reach-1         ,94876
     584     845    1071     674    1345    2684    2152
River Rch & RM=Lytle Creek,Reach-1         ,81295
     934    1387    1786    1141    2277    4544    3756
River Rch & RM=Lytle Creek,Reach-1         ,76774
     966    1430    1838    1172    2338    4665    3838
River Rch & RM=Lytle Creek,Reach-1         ,70093
    1017    1506    1936    1234    2463    4914    4041
River Rch & RM=Lytle Creek,Reach-1         ,66503
    1254    1873    2421    1551    3095    6176    5131
River Rch & RM=Lytle Creek,Reach-1         ,62780
    1360    2034    2632    1688    3368    6720    5592
River Rch & RM=Lytle Creek,Reach-1         ,59952
    1502    2253    2920    1875    3741    7465    6229
River Rch & RM=Lytle Creek,Reach-1         ,58923
    2081    3136    4080    2627    5241   10457    8769
River Rch & RM=Lytle Creek,Reach-1         ,52412
    2533    3836    5008    3234    6452   12874   10856
River Rch & RM=Lytle Creek,Reach-1         ,47505
    2610    3951    5156    3328    6639   13247   11162
River Rch & RM=Lytle Creek,Reach-1         ,43111
    2605    3932    5120    3297    6578   13125   11008
River Rch & RM=Lytle Creek,Reach-1         ,31068
    2739    4129    5373    3457    6898   13762   11520
River Rch & RM=Lytle Creek,Reach-1         ,25857
    2742    4130    5371    3453    6891   13749   11493
River Rch & RM=Lytle Creek,Reach-1         ,21642
    2976    4488    5843    3759    7501   14967   12530
River Rch & RM=Lytle Creek,Reach-1         ,16664
    2964    4460    5797    3724    7430   14825   12370
River Rch & RM=Lytle Creek,Reach-1         ,9206
    3000    4512    5864    3766    7514   14993   12505
River Rch & RM=Lytle Creek,Reach-1         ,8140
    2998    4507    5854    3758    7498   14961   12466
River Rch & RM=Lytle Creek,Reach-1         ,6872
    2942    4407    5711    3657    7297   14560   12072
Boundary for River Rch & Prof#=Lytle Creek,Reach-1         , 1
Up Type= 0
Dn Type= 3
Dn Slope=0.005
Boundary for River Rch & Prof#=Lytle Creek,Reach-1         , 2
Up Type= 0
Dn Type= 3
Dn Slope=0.005
Boundary for River Rch & Prof#=Lytle Creek,Reach-1         , 3
Up Type= 0
Dn Type= 3
Dn Slope=0.005
Boundary for River Rch & Prof#=Lytle Creek,Reach-1         , 4
Up Type= 0
Dn Type= 3
Dn Slope=0.005
Boundary for River Rch & Prof#=Lytle Creek,Reach-1         , 5
Up Type= 0
Dn Type= 3
Dn Slope=0.005
Boundary for River Rch & Prof#=Lytle Creek,Reach-1         , 6
Up Type= 0
Dn Type= 3
Dn Slope=0.005
Boundary for River Rch & Prof#=Lytle Creek,Reach-1         , 7
Up Type= 0
Dn Type= 3
Dn Slope=0.005
DSS Import GetInterval= 0
DSS Import GetPeak= 0
DSS Import FillOption= 0

--- Lytle Creek.g02 (geometry) ---

Geom Title=LytleCr
Program Version=4.10

River Reach=Lytle Creek     ,Reach-1
Reach XY= 30
        1629755.        6790838.      1627115.27      6794587.07
      1624152.71      6795343.06      1623415.83       6796543.7
        1619555.        6796738.      1614975.92       6798801.4
      1614975.47      6800784.73      1613668.54      6801467.32
      1612839.15      6805741.73      1611479.42      6805612.96
      1610897.33      6808994.53      1609596.61        6809358.
      1609591.01      6811110.25      1606495.05      6815073.23
      1604411.21      6815731.98      1605152.76      6817123.51
      1604202.73      6819217.06      1604858.01      6819996.63
      1603614.74      6819981.16      1603987.33       6822147.3
      1602064.68      6823633.74      1601952.32      6827795.59
      1600648.55      6829737.42      1600811.52      6832579.42
      1599533.31      6832355.87      1598960.46      6834996.74
      1598143.39      6834955.85      1596580.79      6837076.55
        1596655.        6840738.        1592055.        6847938.

Type RM Length L Ch R = 1 ,97944   ,139,139,139
BEGIN DESCRIPTION:
Lytle Creek 98308.404
END DESCRIPTION:
XS GIS Cut Line= 3
      1629457.47      6790785.77      1629754.74      6790871.55
      1629996.49      6790925.08
#Sta/Elev= 30
  4690.6 1995.63    4749 1995.06  4781.7 1994.16  4787.9 1993.34  4799.7 1993.08
  4821.5 1992.62  4839.3 1993.29  4875.4 1992.27  4885.8 1990.21    4894 1986.88
  4901.9 1985.11  4904.6 1984.34  4904.8 1983.84  4908.3 1983.84  4908.6 1984.34
  4938.1 1985.24  4948.2 1984.56  4958.6 1985.23  4979.5 1984.45    5006 1985.16
  5011.2 1984.59  5020.7 1984.93  5041.2 1989.31  5049.7  1992.3  5054.8 1993.44
  5092.4 1994.55  5098.4  1996.1  5133.4 1998.68  5207.7 2000.16  5247.6 2000.92
#Mann= 7 ,-1 , 0
  4690.6     .05       0  4799.7     .12       0  4839.3      .1       0
  4901.9     .12       0  4904.6     .07       0  4908.6     .12       0
  5207.7     .05       0
Bank Sta=4904.6,4908.6
XS Rating Curve= 0 ,0
Exp/Cntr=0.3,0.1

Type RM Length L Ch R = 1 ,97805   ,106,106,106
BEGIN DESCRIPTION:
Lytle Creek 98184.62
END DESCRIPTION:
XS GIS Cut Line= 2
      1629385.85      6790926.46      1629945.92      6791048.44
#Sta/Elev= 30
  4681.8 1991.98  4709.5 1992.02    4773 1990.35  4793.5 1990.15    4803 1990.55
  4824.2 1989.16  4834.4 1988.81  4851.7 1988.95  4856.8 1988.62  4865.2 1989.01
  4900.7 1987.89  4916.3 1986.62  4936.8 1986.18  4944.7 1985.39  4949.8 1985.59
  4977.7 1983.22    4986 1983.09  4986.2 1982.59  4989.7 1982.59    4990 1983.09
  4998.9  1983.8  5008.4 1985.35  5028.9 1987.85  5049.4  1991.2  5059.6 1992.14
  5091.9 1993.18    5121 1996.21  5141.5 1997.47  5151.7 1997.31    5255 1999.04
#Mann= 5 ,-1 , 0
  4681.8     .05       0    4803      .1       0    4986     .07       0
    4990      .1       0  5059.6     .05       0
Bank Sta=4986,4990
XS Rating Curve= 0 ,0
Exp/Cntr=0.3,0.1

Type RM Length L Ch R = 1 ,97699   ,185,185,185
BEGIN DESCRIPTION:
Lytle Creek 98062.36
END DESCRIPTION:
XS GIS Cut Line= 3
      1629403.05      6790954.42       1629621.5      6791069.62
      1629840.98       6791207.2
#Sta/Elev= 30
  4729.7 1991.51  4764.9 1991.24  4770.5 1992.27  4777.1 1990.95  4792.5 1990.85
  4799.7 1989.89  4808.9 1990.03    4821  1989.4    4845 1988.56    4853 1988.88
  4858.6 1987.46    4875 1987.64  4912.8 1986.83  4935.4 1985.57  4946.7 1984.17
  4955.3 1984.19  4984.9 1984.06  4998.2 1980.76  4998.4 1980.26  5001.9 1980.26
  5002.2 1980.76  5006.1 1981.63  5015.5 1985.41  5036.7 1987.96  5051.6 1988.32
  5073.2 1990.24    5087 1990.44  5115.7    1992  5152.2 1995.07  5235.7 1995.82
#Mann= 5 ,-1 , 0
  4729.7     .05       0    4821      .1       0  4955.3     .05       0
  4998.2     .05       0  5002.2     .05       0
Bank Sta=4998.2,5002.2
XS Rating Curve= 0 ,0
Exp/Cntr=0.3,0.1

Type RM Length L Ch R = 1 ,97514   ,214,214,214
BEGIN DESCRIPTION:
Mapping XS cb8f6ab7
END DESCRIPTION:
XS GIS Cut Line= 4
      1629332.16      6790936.41      1629437.68       6791025.6
      1629523.83      6791262.77      1629713.95      6791346.39
#Sta/Elev= 30
  4731.7 1992.85  4770.5  1991.9  4834.2 1991.87  4840.8 1990.65  4848.5 1990.74
  4855.1 1988.54  4862.8 1988.61  4867.9 1987.27  4912.7 1986.09  4933.1 1985.09
  4938.4 1985.46  4957.5  1983.7  4963.7 1981.97  4978.8 1981.59  4986.9 1978.76
  4987.2 1978.26  4990.8 1978.26  4991.1 1978.76  4994.3  1978.9  5000.1 1981.51
  5010.7 1983.58    5032 1983.11  5074.6 1983.79  5111.4 1985.81    5117 1986.75
  5167.1 1987.95  5224.7 1990.63  5242.6 1990.73  5318.1 1994.57  5329.9 1994.72
#Mann= 5 ,-1 , 0
  4731.7     .05       0  4912.7      .1       0  4938.4     .05       0
  4986.9     .05       0  4991.1     .05       0
Bank Sta=4986.9,4991.1
XS Rating Curve= 0 ,0
Exp/Cntr=0.3,0.1

Type RM Length L Ch R = 1 ,97300   ,243,243,243
BEGIN DESCRIPTION:
Lytle Creek 97631.83
END DESCRIPTION:
XS GIS Cut Line= 2
      1629120.45      6790984.32      1629468.03      6791464.65
#Sta/Elev= 30
  4731.2 1994.31  4759.4 1995.88  4772.8 1995.49  4780.3 1994.13    4795 1993.84
  4830.5 1991.33  4851.4    1991  4916.4 1987.79  4922.6 1988.09  4945.6 1987.21
    4952  1986.1  4958.1 1986.24  4972.8 1984.61  4987.5 1980.66  4992.9 1977.66
  4993.2 1977.16  4996.8 1977.16  4997.1 1977.66  5002.2 1978.09  5008.4 1979.97
  5023.1 1980.67  5073.4  1980.7  5123.7 1982.29  5138.4 1984.36  5167.8 1985.47
  5217.1 1988.67  5224.2  1989.9  5230.4 1992.45  5238.9 1991.27  5324.1 1993.76
#Mann= 3 ,-1 , 0
  4731.2     .05       0  4992.9     .05       0  4997.1     .05       0
Bank Sta=4992.9,4997.1
XS Rating Curve= 0 ,0
Exp/Cntr=0.3,0.1

Type RM Length L Ch R = 1 ,97057   ,322,322,322
BEGIN DESCRIPTION:
Lytle Creek 97411.86
END DESCRIPTION:
XS GIS Cut Line= 2
      1628909.55      6791130.53      1629298.36      6791608.19
#Sta/Elev= 30
    4703 1989.62  4719.3 1988.93  4740.1  1989.3  4783.2 1988.81  4797.6 1987.51
  4804.1  1987.9  4832.8 1986.73  4861.5 1984.03  4882.3 1983.37  4890.3 1982.21
  4925.4 1979.81  4982.9 1978.55  4989.4 1976.93  4994.2 1974.53  4994.5 1974.03
  4998.1 1974.03  4998.5 1974.53  5018.1 1978.31  5067.6 1978.41    5082 1978.93
  5102.8 1981.15  5110.7 1981.39  5117.2 1982.65  5145.9 1983.17  5160.3 1984.92
  5166.7 1986.43  5195.5  1989.9  5252.9 1991.59  5259.4 1992.21  5318.9 1993.55
#Mann= 3 ,-1 , 0
    4703     .05       0  4994.2     .05       0  4998.5     .05       0
Bank Sta=4994.2,4998.5
XS Rating Curve= 0 ,0
Exp/Cntr=0.3,0.1

Type RM Length L Ch R = 1 ,96735   ,252,252,252
BEGIN DESCRIPTION:
Lytle Creek 97066.38
END DESCRIPTION:
XS GIS Cut Line= 3
      1628640.03      6791400.24      1628845.72      6791544.75
      1629180.15      6791747.75
#Sta/Elev= 30
  4769.7 1987.93    4793 1987.42  4807.8 1985.61  4864.5 1982.86    4915 1978.17
  4944.6 1976.81  4950.7 1975.73  4965.5 1975.82  4971.6 1975.36  4980.3 1975.91
    4993 1971.66  4993.3 1971.16  4996.9 1971.16  4997.3 1971.66  5001.3 1971.66
    5008 1973.58  5016.1  1974.7  5031.5 1974.56  5074.2 1975.24    5080 1975.75
  5089.7 1975.57  5095.5 1977.48    5111 1977.61  5132.4 1978.83  5160.6 1982.98
  5190.5 1985.04  5233.2 1985.95  5264.1 1987.82  5312.7 1989.69  5412.3 1992.84
#Mann= 3 ,-1 , 0
  4769.7     .05       0    4993     .05       0  4997.3     .05       0
Bank Sta=4993,4997.3
XS Rating Curve= 0 ,0
Exp/Cntr=0.3,0.1

Type RM Length L Ch R = 1 ,96483   ,224,224,224
BEGIN DESCRIPTION:
Lytle Creek 96796.09
END DESCRIPTION:
XS GIS Cut Line= 3
      1628317.03       6791704.9      1628755.88      6791770.01
      1629150.85      6791857.06
#Sta/Elev= 30
    4542 1982.03  4730.2 1982.26  4772.5 1981.75  4833.1 1980.06  4903.9 1979.33
  4938.6 1978.16  4974.7 1972.66  4982.7 1970.89  4987.8 1970.89  4992.5 1970.02
  4992.9 1969.52  4996.5 1969.52  4996.9 1970.02  5005.2  1970.2  5025.7 1972.18
  5048.7 1972.93  5087.2  1976.1  5092.4 1977.12  5097.5  1977.1  5107.6 1978.76
  5136.1 1980.07  5141.2 1979.86  5148.6 1980.73  5179.3 1982.37  5184.9 1983.25
    5210 1984.86  5233.7 1985.75  5277.5 1988.79  5326.3 1989.93  5390.1 1993.05
#Mann= 3 ,-1 , 0
    4542     .05       0  4992.5     .05       0  4996.9     .05       0
Bank Sta=4992.5,4996.9
XS Rating Curve= 0 ,0
Exp/Cntr=0.3,0.1

Type RM Length L Ch R = 1 ,96259   ,138,138,138
BEGIN DESCRIPTION:
Lytle Creek 96542.94
END DESCRIPTION:
XS GIS Cut Line= 3
      1628363.33      6791912.45      1628757.88      6791991.89
      1629109.48      6792046.58
#Sta/Elev= 30
  4575.7 1979.65  4677.1 1979.88  4829.6  1976.8  4873.2 1976.48  4880.4 1977.16
  4893.6 1976.94  4924.2  1974.4  4931.2 1972.75  4936.3 1972.67  4954.8 1969.54
  4978.2 1967.72  4980.7  1966.7  4981.1  1966.2  4984.7  1966.2  4985.1  1966.7
  4987.9 1967.36  4995.5 1966.96  5005.6 1967.52  5015.7 1969.04    5036 1974.22
  5045.8 1975.34  5113.7 1978.56  5118.8  1978.1  5181.7 1981.04    5208 1983.91
  5238.4 1984.84  5244.5  1985.8  5268.7 1987.41  5307.4 1991.25    5334 1992.53
#Mann= 3 ,-1 , 0
  4575.7     .05       0  4980.7     .05       0  4985.1     .05       0
Bank Sta=4980.7,4985.1
XS Rating Curve= 0 ,0
Exp/Cntr=0.3,0.1

Type RM Length L Ch R = 1 ,96121   ,74,74,74
BEGIN DESCRIPTION:
Lytle Creek 96407
END DESCRIPTION:
XS GIS Cut Line= 3
      1628391.69      6792093.01      1628725.93      6792118.19
      1629008.01      6792133.81
#Sta/Elev= 30
  4665.3 1976.88  4728.8 1977.17    4789 1976.92  4869.2 1975.56  4909.3 1974.16
  4919.3 1974.35  4927.9 1974.12  4939.4 1973.11  4959.4 1972.16  4979.5 1968.26
  4989.5 1966.61  4995.3  1966.5  4995.7    1966  4999.3    1966  4999.7  1966.5
  5009.6 1966.51  5019.6 1967.03  5029.6 1968.54  5039.6  1970.7  5059.7 1972.58
  5069.7 1973.16  5091.1  1973.7  5149.8 1977.07  5179.8 1978.36  5239.9 1982.64
    5260 1983.57  5266.7 1984.19  5271.7 1984.09    5279 1984.88    5283 1984.88
#Mann= 3 ,-1 , 0
  4665.3     .05       0  4995.3     .05       0  4999.7     .05       0
Bank Sta=4995.3,4999.7
XS Rating Curve= 0 ,0
Exp/Cntr=0.3,0.1

Type RM Length L Ch R = 1 ,96047   ,195,195,195
BEGIN DESCRIPTION:
Lytle Creek 96332.97
END DESCRIPTION:
XS GIS Cut Line= 3
      1628314.45      6792168.53      1628700.76       6792185.9
       1629067.1      6792216.28
#Sta/Elev= 30
  4614.2  1975.3  4804.9 1976.27    4885 1974.93  4915.1 1974.89  4938.2 1974.08
  4955.1 1972.62  4975.1 1968.01  4985.1 1966.57  4992.9 1966.41  4993.3 1965.91
  4996.9 1965.91  4997.3 1966.41  5000.5 1967.21  5005.5 1967.21  5015.2 1968.31
  5045.3 1970.28  5065.4 1971.07  5083.6 1973.01  5088.7 1973.05  5095.5 1974.15
  5105.5 1974.79  5135.6 1975.94  5185.8 1978.65  5204.3 1979.77  5209.3 1980.93
    5246 1982.69  5266.1 1983.15  5286.1 1984.67  5306.2 1985.52  5368.5 1989.65
#Mann= 3 ,-1 , 0
  4614.2     .05       0  4992.9     .05       0  4997.3     .05       0
Bank Sta=4992.9,4997.3
XS Rating Curve= 0 ,0
Exp/Cntr=0.3,0.1

Type RM Length L Ch R = 1 ,95852   ,73,73,73
BEGIN DESCRIPTION:
Lytle Creek 96131.29
END DESCRIPTION:
XS GIS Cut Line= 3
      1628334.04      6792282.35      1628653.45      6792372.61
       1628986.1      6792482.34
#Sta/Elev= 30
  4679.2 1973.87  4751.4 1974.45  4815.3 1973.86  4868.9    1972  4936.9 1970.68
  4960.8 1969.41  4976.1 1966.48  5000.1  1965.9  5000.5  1965.4  5004.1  1965.4
  5004.5  1965.9  5015.2 1966.16  5023.3 1967.92  5041.7 1970.68  5073.4 1972.55
  5086.5 1972.53  5128.6 1974.05  5136.9 1975.11  5142.2  1974.8  5168.7 1977.17
    5174 1976.85  5181.2 1978.17  5200.5 1979.63  5205.7 1979.23  5232.2 1982.44
  5237.5 1982.51  5244.4 1983.79    5276 1985.25  5318.1 1985.93  5361.4 1987.66
#Mann= 3 ,-1 , 0
  4679.2     .05       0  5000.1     .05       0  5004.5     .05       0
Bank Sta=5000.1,5004.5
XS Rating Curve= 0 ,0
Exp/Cntr=0.3,0.1

Type RM Length L Ch R = 1 ,95779   ,168,168,168
BEGIN DESCRIPTION:
Mapping XS f53f254b
END DESCRIPTION:
XS GIS Cut Line= 5
      1628358.85      6792320.09      1628525.52      6792370.44
      1628650.52      6792465.92      1628782.46      6792655.16
      1628964.72      6792738.48
#Sta/Elev= 30
  4745.6 1973.39  4789.4 1974.09    4846 1973.16  4866.9 1972.09  4921.8 1971.05
  4924.6 1970.36  4953.7 1969.79    4989  1965.9  5001.4 1965.52  5001.8 1965.02
  5005.4 1965.02  5005.8 1965.52  5089.6 1966.22  5140.2 1965.63  5161.1 1966.27
  5167.2 1967.99  5182.1 1970.31    5203 1972.83  5211.8 1972.99  5225.8  1974.6
  5238.8  1977.8  5274.6 1981.31  5349.8 1984.33  5372.8 1985.05  5378.3 1984.76
  5418.9 1986.73  5447.4 1987.08  5493.4 1988.94  5498.9 1988.29  5508.1  1988.6
#Mann= 3 ,-1 , 0
  4745.6     .05       0  5001.4     .05       0  5005.8     .05       0
Bank Sta=5001.4,5005.8
XS Rating Curve= 0 ,0
Exp/Cntr=0.3,0.1

Type RM Length L Ch R = 1 ,95611   ,246,246,246
BEGIN DESCRIPTION:
Lytle Creek 95878
END DESCRIPTION:
XS GIS Cut Line= 3
      1628343.74      6792375.31      1628463.13      6792528.34
      1628606.36      6792816.97
#Sta/Elev= 30
    4833 1972.73  4857.4 1972.38  4863.8 1972.56  4921.7  1970.6    4928 1970.07
  4942.5 1969.63  4956.9 1968.46  4963.3 1968.37  4977.7 1967.44    4998 1965.23
  4998.5 1964.73  5002.2 1964.73  5002.7 1965.23  5006.7 1966.24    5014 1966.95
  5037.4 1967.02  5071.4 1967.76    5116 1970.23  5138.3 1971.14  5149.5  1971.2
  5183.1 1972.97  5194.2 1973.23  5205.5 1974.02  5216.5 1974.25  5227.9 1975.09
  5244.7 1975.33  5289.5 1977.95  5295.1 1977.64  5328.1 1978.76  5349.3  1979.8
#Mann= 3 ,-1 , 0
    4833     .05       0    4998     .05       0  5002.7     .05       0
Bank Sta=4998,5002.7
XS Rating Curve= 0 ,0
Exp/Cntr=0.3,0.1

Type RM Length L Ch R = 1 ,95365   ,190,190,190
BEGIN DESCRIPTION:
Lytle Creek 95633.92
END DESCRIPTION:
XS GIS Cut Line= 3
      1628068.69      6792412.78      1628257.47      6792642.78
      1628554.79      6792916.23
#Sta/Elev= 30
  4703.3 1969.04  4733.2 1968.62  4774.8 1969.04  4782.7 1968.79  4817.9 1969.34
  4881.7  1969.3    4904 1968.39    4917 1968.28  4924.8 1967.36  4945.6  1965.8
  4967.8 1965.12  4974.3 1964.32  4986.3 1961.85  4986.8 1961.35  4990.5 1961.35
    4991 1961.85  5000.9 1962.25  5010.1 1963.31  5016.9 1964.67  5031.1  1964.9
  5059.5 1966.18  5066.2 1967.29  5080.4 1968.52  5087.8 1968.79  5094.6 1969.59
    5123 1970.67  5236.4  1977.6  5299.9 1980.07  5356.6 1980.52  5404.8 1981.97
#Mann= 3 ,-1 , 0
  4703.3     .05       0  4986.3     .05       0    4991     .05       0
Bank Sta=4986.3,4991
XS Rating Curve= 0 ,0
Exp/Cntr=0.3,0.1

Type RM Length L Ch R = 1 ,95175   ,299,299,299
BEGIN DESCRIPTION:
Mapping XS 38325b7c
END DESCRIPTION:
XS GIS Cut Line= 4
      1627923.27      6792338.96      1628003.08      6792656.72
      1628242.29      6792889.69      1628550.24      6792949.24
#Sta/Elev= 30
    4513 1971.17  4553.3  1970.4  4635.7  1967.8    4677 1967.07  4871.2 1965.52
  4934.8 1964.62  4977.3 1963.35  4984.3 1962.12  4996.1 1961.16  4996.6 1960.66
  5000.3 1960.66  5000.8 1961.16  5012.5 1963.64  5019.7 1964.63  5033.9 1965.38
    5055 1967.51  5076.3 1968.37  5097.4 1967.85  5125.7 1968.16  5178.5  1969.9
  5228.2 1973.24  5244.1 1974.93  5258.8 1975.94    5269 1976.04  5289.3 1977.47
  5295.9 1978.34  5330.1    1980    5381 1981.12  5442.1 1981.54  5488.2 1982.44
#Mann= 3 ,-1 , 0
    4513     .05       0  4996.1     .03       0  5000.8     .05       0
Bank Sta=4996.1,5000.8
XS Rating Curve= 0 ,0
Exp/Cntr=0.3,0.1

Type RM Length L Ch R = 1 ,94876   ,233,233,233
BEGIN DESCRIPTION:
Lytle Creek 95413.9
END DESCRIPTION:
XS GIS Cut Line= 4
      1627348.95      6792821.16      1627675.96      6792874.85
      1628032.09      6793039.06      1628561.67      6793083.56
#Sta/Elev= 30
  4410.7 1981.42  4447.2 1980.47  4558.7  1973.3  4589.1  1972.6  4619.5 1970.99
    4660 1969.63    4811 1967.01  4833.9 1965.25  4840.1 1964.33  4851.1 1963.94
  4862.4 1962.87  4873.2 1964.08  4885.3 1964.56  4971.6 1963.84  4994.3 1961.48
  5003.2 1960.06  5003.7 1959.56  5007.4 1959.56    5008 1960.06    5023 1962.74
  5060.4 1964.24  5068.9 1965.19  5097.4 1964.68  5337.9 1970.32  5421.7 1973.64
  5448.3 1975.96  5536.6 1979.41  5558.7 1979.69  5598.8 1981.48  5665.7 1983.31
#Mann= 3 ,-1 , 0
  4410.7     .05       0  5003.2     .05       0    5008     .05       0
Bank Sta=5003.2,5008
XS Rating Curve= 0 ,0
Exp/Cntr=0.3,0.1

Type RM Length L Ch R = 1 ,94643   ,169,169,169
BEGIN DESCRIPTION:
Mapping XS 04d59858
END DESCRIPTION:
XS GIS Cut Line= 4
      1627129.91      6793054.75      1627670.27      6793119.86
      1628245.35      6793152.41      1628618.64      6793182.79
#Sta/Elev= 30
    4372 1982.74  4417.4 1980.79  4487.9 1979.25  4548.4 1975.98  4578.6 1975.88
  4628.9 1973.96  4649.1 1973.56  4669.2 1975.27  4719.6 1974.21  4780.2 1969.14
  4890.8 1964.92    4911 1962.83  4916.1 1961.45  4921.1 1961.45  4951.1 1956.82
  4965.4 1956.57  4966.5 1956.07  4972.5 1956.57    4974  1957.4  5001.1 1958.99
  5021.2 1962.24  5081.3 1962.76  5121.3 1961.57  5271.6 1964.41  5451.9 1968.94
  5572.2 1972.95  5612.3 1976.38  5625.1 1976.07  5792.9 1983.43  5866.8 1985.61
#Mann= 3 ,-1 , 0
    4372     .05       0  4965.4     .05       0  4972.5     .05       0
Bank Sta=4965.4,4972.5
XS Rating Curve= 0 ,0
Exp/Cntr=0.3,0.1

Type RM Length L Ch R = 1 ,94474   ,185,185,185
BEGIN DESCRIPTION:
Mapping XS 56ed5623
END DESCRIPTION:
XS GIS Cut Line= 4
      1627092.17      6793168.04      1627362.98      6793254.84
      1627928.95       6793291.3      1628609.52      6793230.53
#Sta/Elev= 30
  4371.1 1982.22  4452.9 1980.01  4468.6 1978.75  4479.1 1979.25  4517.1 1976.99
  4542.1 1976.59  4594.6 1973.75  4707.6 1970.73  4837.9 1964.85  4867.9 1964.87
  4968.2  1963.2  4988.2  1959.7  4994.7 1959.15  4995.8 1958.65  5000.7 1958.65
  5001.8 1959.15  5008.2 1961.16  5138.5 1961.14  5178.6 1962.44  5188.6 1961.88
  5228.7 1961.74    5299 1963.78  5529.9 1968.52  5630.3 1972.07  5654.3 1973.36
  5680.5 1976.25  5765.8 1979.62  5831.1 1983.43  5877.2 1985.13  5905.9 1985.44
#Mann= 3 ,-1 , 0
  4371.1     .05       0  4994.7     .05       0  5001.8     .05       0
Bank Sta=4994.7,5001.8
XS Rating Curve= 0 ,0
Exp/Cntr=0.3,0.1

Type RM Length L Ch R = 1 ,94289   ,174,174,174
BEGIN DESCRIPTION:
Lytle Creek 94789.65
END DESCRIPTION:
XS GIS Cut Line= 3
      1627100.25      6793434.09      1627536.24      6793468.46
      1628597.77      6793379.41
#Sta/Elev= 30
    4330 1978.34  4475.2 1971.06  4555.4 1969.46  4595.6 1967.85  4645.7 1966.74
  4699.4 1964.41  4764.2  1962.9  4786.2 1963.01    4832 1961.64  4966.8 1960.87
  4976.8 1960.57  4993.3 1957.89  4994.5 1957.39  4999.4 1957.39  5000.5 1957.89
  5006.9 1957.91    5017 1959.55    5037 1959.28    5067 1960.56  5127.4 1960.95
  5192.1 1962.07  5227.7 1963.27    5298 1963.86  5398.3 1965.88  5418.4 1965.76
  5518.7 1969.31  5649.2 1976.78  5679.3 1977.41  5719.4 1979.42  5832.6 1983.05
#Mann= 3 ,-1 , 0
    4330     .05       0  4993.3     .05       0  5000.5     .05       0
Bank Sta=4993.3,5000.5
XS Rating Curve= 0 ,0
Exp/Cntr=0.3,0.1

Type RM Length L Ch R = 1 ,94115   ,171,171,171
BEGIN DESCRIPTION:
Lytle Creek 94361.14
END DESCRIPTION:
XS GIS Cut Line= 3
      1627055.58      6793588.28      1627806.43      6793612.15
       1628780.4      6793575.27
#Sta/Elev= 30
    4224  1976.1  4283.5  1973.8  4343.5 1972.79  4453.5 1967.58  4483.6  1967.1
  4563.6 1964.49  4623.6 1963.24  4673.7 1963.91  4743.7  1960.7  4753.7 1959.81
  4793.7 1959.58  4813.7 1960.22  4863.7 1960.35  5000.2 1958.73  5001.3 1958.23
  5006.3 1958.23  5007.5 1958.73  5013.8  1959.6  5053.9  1959.9  5163.9 1964.03
    5234  1964.7  5444.1 1969.73  5534.2 1973.04  5604.3 1976.59  5614.3 1976.32
  5644.3 1978.11  5714.3  1981.1  5747.5 1981.38  5914.5 1986.99  5949.9 1988.62
#Mann= 3 ,-1 , 0
    4224     .05       0  5000.2     .05       0  5007.5     .05       0
Bank Sta=5000.2,5007.5
XS Rating Curve= 0 ,0
Exp/Cntr=0.3,0.1

Type RM Length L Ch R = 1 ,93944   ,379,379,379
BEGIN DESCRIPTION:
Lytle Creek 94191.93
END DESCRIPTION:
XS GIS Cut Line= 3
      1626927.48      6793792.27      1627754.35      6793766.23
      1628756.92      6793748.87
#Sta/Elev= 30
  4161.3 1974.65  4188.8  1974.2  4218.8 1971.43  4378.9 1965.32    4449 1963.76
    4469 1964.31    4539 1961.87  4679.1 1961.37  4709.1 1959.74  4789.1 1958.16
  4959.2 1958.73  4995.6  1957.4  4996.7  1956.9  5002.9  1957.4  5039.2 1961.81
  5069.2 1964.34  5109.2 1962.25  5129.3 1962.35  5449.3  1968.1  5529.3 1972.47
  5549.3 1972.49  5609.3 1975.33  5649.3 1978.74  5659.3 1977.67  5669.3 1977.95
  5769.3 1984.28  5879.4 1987.89  5889.4 1989.26  5909.4 1988.72  5991.3 1990.83
#Mann= 3 ,-1 , 0
  4161.3     .05       0  4995.6     .05       0  5002.9     .05       0
Bank Sta=4995.6,5002.9
XS Rating Curve= 0 ,0
Exp/Cntr=0.3,0.1

Type RM Length L Ch R = 1 ,93565   ,412,412,412
BEGIN DESCRIPTION:
Lytle Creek 93802.39
END DESCRIPTION:
XS GIS Cut Line= 3
      1626982.18      6793961.02       1627755.6      6794125.08
      1628487.35      6794119.87
#Sta/Elev= 30
  4222.4 1965.53  4337.7 1961.17  4480.8 1957.67  4667.8  1957.1  4712.4 1958.89
  4746.6 1957.51  4811.7 1956.91  4838.6 1953.49  4856.2    1956  4889.7 1957.07
  4971.5 1956.97  4996.3 1953.11  4997.5 1952.61  5003.7 1953.11  5010.2 1957.22
  5062.4 1959.39  5202.4 1963.22  5282.4 1964.32  5301.4 1965.13  5312.4 1967.64
  5352.4 1969.21  5382.4 1968.99  5412.4 1970.56  5472.4  1970.5  5482.4 1970.95
  5502.4 1974.57  5552.4 1975.95  5562.4 1977.31  5592.4 1976.34  5744.8  1983.5
#Mann= 3 ,-1 , 0
  4222.4     .05       0  4996.3     .05       0  5003.7     .05       0
Bank Sta=4996.3,5003.7
XS Rating Curve= 0 ,0
Exp/Cntr=0.3,0.1

Type RM Length L Ch R = 1 ,93153   ,310,310,310
BEGIN DESCRIPTION:
Lytle Creek 93421.23
END DESCRIPTION:
XS GIS Cut Line= 3
      1626906.69      6794044.37      1627487.38      6794359.46
      1628049.86      6794658.93
#Sta/Elev= 30
  4369.2 1964.43    4555 1959.41  4620.6 1959.71  4718.5 1957.11  4871.6 1955.07
  4937.1 1955.91    4959 1953.45  4969.5  1954.3  4981.7 1949.54  4993.3 1949.05
  4994.5 1948.55  5000.7 1949.05  5013.2 1949.84  5025.7 1955.12  5151.8 1955.97
  5210.9 1955.11    5337 1962.34  5389.7 1961.78  5397.3 1963.53  5419.2 1965.41
  5468.3 1967.48  5507.1 1965.75  5559.6 1967.35  5589.3 1969.79  5619.9 1970.22
  5633.2 1971.04  5649.5 1977.75  5655.2 1977.41  5661.5 1980.42  5667.1 1980.42
#Mann= 5 ,-1 , 0
  4369.2     .05       0  4993.3     .05       0  5000.7     .05       0
  5468.3     .12       0  5619.9     .05       0
Bank Sta=4993.3,5000.7
XS Rating Curve= 0 ,0
Exp/Cntr=0.3,0.1

Type RM Length L Ch R = 1 ,92843   ,500,500,500
BEGIN DESCRIPTION:
Lytle Creek 93090.31
END DESCRIPTION:
XS GIS Cut Line= 3
      1626890.99        6794099.      1627216.54      6794531.33
      1628018.64      6795015.71
#Sta/Elev= 30
  4468.7 1962.55  4520.3 1961.54  4564.1  1957.8  4584.9 1959.28  4599.5 1956.95
    4614 1956.54  4628.6 1956.77  4642.7 1958.92  4670.3 1960.52  4784.8 1960.08
    4893 1956.41  4949.3 1955.68    4993 1952.22  4995.5 1950.06  4996.6 1949.56
    5003 1950.06    5029 1953.03  5078.2 1954.06  5151.3 1954.49    5160 1952.45
    5195 1954.63  5253.4  1953.4  5421.1 1954.95  5712.2 1962.58  5727.7 1963.98
  5779.1 1965.21  5785.9    1967  5801.4 1967.64  5822.8 1964.54  5946.9 1966.98
#Mann= 3 ,-1 , 0
  4468.7     .05       0  4995.5     .05       0    5003     .05       0
Bank Sta=4995.5,5003
XS Rating Curve= 0 ,0
Exp/Cntr=0.3,0.1

Type RM Length L Ch R = 1 ,92343   ,519,519,519
BEGIN DESCRIPTION:
Lytle Creek 92595.09
END DESCRIPTION:
XS GIS Cut Line= 4
      1626668.15       6794157.2      1626760.37      6794646.33
      1626944.71      6795006.11      1626979.71      6795053.35
#Sta/Elev= 30
  4495.7 1964.29  4508.7 1964.16    4527 1962.63  4556.1 1962.75  4561.2 1962.08
  4608.5 1960.63  4613.6    1960  4723.5 1957.16  4730.6 1955.71  4750.9 1954.43
  4791.6 1949.67  4974.8  1950.5    4985  1949.8  4990.8 1947.02  5002.8 1946.72
    5004 1946.22  5009.2 1946.22  5010.3 1946.72  5013.4 1948.12    5029 1950.77
    5080 1949.91  5146.6  1949.8  5197.6 1950.47  5207.6 1950.08  5235.4 1951.09
    5252 1950.33  5318.6 1949.94    5402 1950.33  5427.3 1951.31  5456.5 1951.33
#Mann= 3 ,-1 , 0
  4495.7     .05       0  5002.8     .05       0  5010.3     .05       0
Bank Sta=5002.8,5010.3
XS Rating Curve= 0 ,0
Exp/Cntr=0.3,0.1

Type RM Length L Ch R = 1 ,91824   ,473,473,473
BEGIN DESCRIPTION:
Lytle Creek 92056
END DESCRIPTION:
XS GIS Cut Line= 3
      1626238.39      6794123.56      1626263.78      6794857.45
      1626510.57      6795152.25
#Sta/Elev= 30
  4387.1 1965.75  4430.1  1964.9  4435.1 1965.65  4511.6 1961.83  4531.6 1959.87
  4551.6 1960.68  4571.7 1958.69  4631.7 1955.84  4711.7 1952.78  4724.8 1953.15
  4841.8 1947.83  4871.8 1947.55  4891.8  1946.1  4911.9 1947.17  4941.9 1943.78
  4951.9 1943.72  4961.9 1945.44  4971.9 1942.78  4991.9 1942.87  4998.1  1942.2
  4999.3  1941.7  5005.7  1942.2  5021.9 1942.93  5041.9 1945.17    5092 1944.53
  5119.2 1947.33  5125.1 1947.33  5129.9 1946.18  5335.5 1947.74  5505.9 1947.48
#Mann= 3 ,-1 , 0
  4387.1     .05       0  4998.1     .03       0  5005.7     .05       0
Bank Sta=4998.1,5005.7
XS Rating Curve= 0 ,0
Exp/Cntr=0.3,0.1

Type RM Length L Ch R = 1 ,91351   ,460,460,460
BEGIN DESCRIPTION:
Mapping XS 2f5a3b62
END DESCRIPTION:
XS GIS Cut Line= 4
      1625730.16      6793971.84      1625842.14       6794378.1
      1625857.77      6794823.42      1626081.71      6795174.95
#Sta/Elev= 30
  4406.7 1954.13  4515.3 1951.59    4634 1950.65  4702.7 1948.89  4724.3 1949.92
  4742.3 1948.74  4796.9 1947.95    4868 1944.27  4928.1 1943.48  4938.1 1941.39
  4948.1 1940.31  4968.1 1943.42  4978.1 1941.78  4984.3  1937.1  4985.5  1936.6
  4991.9  1937.1  5028.1 1940.71  5038.1 1942.54  5047.7 1942.18  5052.7 1942.79
  5058.1 1941.75  5078.2 1942.92  5148.2 1942.48  5188.2 1942.77  5218.2 1943.86
  5248.3 1942.82  5281.5 1943.14  5317.9 1942.31  5369.5 1942.26  5690.5 1944.65
#Mann= 3 ,-1 , 0
  4406.7     .05       0  4984.3     .05       0  4991.9     .05       0
Bank Sta=4984.3,4991.9
XS Rating Curve= 0 ,0
Exp/Cntr=0.3,0.1

Type RM Length L Ch R = 1 ,90891   ,516,516,516
BEGIN DESCRIPTION:
Mapping XS 617cf102
END DESCRIPTION:
XS GIS Cut Line= 4
      1625406.98      6794489.31      1625516.62      6794698.42
      1625870.79      6795109.87      1626091.08      6795296.47
#Sta/Elev= 30
  4609.2 1946.53  4614.5 1945.99  4620.2 1946.35  4630.3 1944.38  4636.6 1941.75
  4642.2  1942.1  4652.9 1940.71  4658.7  1940.4  4686.8 1940.54  4702.8 1940.05
  4754.5 1939.82  4768.9 1940.22  4835.1 1940.71  4842.3 1941.12    4886 1941.17
  4893.7 1941.54  4943.1 1941.85  4950.3 1941.43  4978.2 1941.62  4996.3 1936.02
  4997.5 1935.52  5002.8 1935.52  5003.9 1936.02    5021 1940.97  5028.7 1941.88
  5042.7 1941.29  5198.7 1941.65  5474.7 1943.63  5531.8 1944.37  5676.9 1945.13
#Mann= 3 ,-1 , 0
  4609.2     .05       0  4996.3     .05       0  5003.9     .05       0
Bank Sta=4996.3,5003.9
XS Rating Curve= 0 ,0
Exp/Cntr=0.3,0.1

Type RM Length L Ch R = 1 ,90375   ,255,255,255
BEGIN DESCRIPTION:
Lytle Creek 90738.38
END DESCRIPTION:
XS GIS Cut Line= 4
       1624912.4      6794426.55      1625145.59      6794800.01
      1625351.17      6795050.62      1625614.99      6795248.66
#Sta/Elev= 30
  4301.3 1941.98  4385.4 1941.21  4427.9 1940.16  4456.3 1940.81  4479.8 1939.61
  4595.4 1939.04  4622.5 1939.71  4631.9 1939.12  4775.7 1938.77  4860.4 1937.49
  4881.3 1935.01  4889.1 1935.03  4895.6 1937.59  4924.3  1938.4  4967.3 1938.18
  4973.8 1938.79  4981.7 1937.72    4996 1934.45  4998.5 1933.37  4999.7 1932.87
  5005.2 1932.87  5006.4 1933.37  5010.4 1937.34  5016.8 1938.01  5023.5 1940.17
  5045.5    1939  5081.6 1939.59  5108.6 1939.13  5195.6 1940.67  5395.6 1942.14
#Mann= 3 ,-1 , 0
  4301.3     .05       0  4998.5     .03       0  5006.4     .05       0
Bank Sta=4998.5,5006.4
XS Rating Curve= 0 ,0
Exp/Cntr=0.3,0.1

Type RM Length L Ch R = 1 ,90120   ,223,223,223
BEGIN DESCRIPTION:
Lytle Creek 90470.76
END DESCRIPTION:
XS GIS Cut Line= 5
      1624834.27      6794506.42       1625033.3       6794896.5
      1625109.28      6795042.61      1625183.45      6795241.12
      1625375.95      6795506.42
#Sta/Elev= 30
  4430.4 1940.35  4440.4    1940  4454.6 1940.76  4512.7 1939.17  4551.5 1939.39
  4640.4 1938.23  4668.3 1938.56  4679.2 1938.06  4735.3 1937.82    4796 1938.04
  4857.1 1937.17  4915.1 1937.42  4937.6 1936.54  4960.2 1936.59  4967.7 1936.37
  4973.3 1935.54  4982.7 1935.46  4989.8 1933.82  4991.5 1930.84  4992.7 1930.34
  4998.2 1930.34  4999.4 1930.84  5005.3 1933.35  5011.9 1934.23  5017.5  1936.1
  5089.5  1936.8  5113.5 1937.84  5144.8 1937.03  5198.9 1937.96  5572.7 1939.37
#Mann= 3 ,-1 , 0
  4430.4     .05       0  4991.5     .05       0  4999.4     .05       0
Bank Sta=4991.5,4999.4
XS Rating Curve= 0 ,0
Exp/Cntr=0.3,0.1

Type RM Length L Ch R = 1 ,89897   ,371,371,371
BEGIN DESCRIPTION:
Lytle Creek 90266.99
END DESCRIPTION:
XS GIS Cut Line= 5
      1624795.56       6794552.1      1624910.04      6794949.07
      1624943.61      6795150.42      1625037.42      6795439.85
      1625303.95      6795524.92
#Sta/Elev= 30
  4351.1 1939.67  4648.6 1936.68  4732.6 1936.92  4752.7 1936.23  4773.3 1936.85
  4826.9 1933.86  4864.5 1934.22  4887.8 1933.65  4905.1 1934.79  4925.4 1934.25
  4968.4 1935.16  4976.3 1934.88  4985.3  1933.1  4990.6 1932.93  4993.4 1931.41
  4994.6 1930.91  5000.1 1930.91  5001.3 1931.41  5022.6 1934.77  5028.9 1936.43
  5054.6  1937.2    5113 1936.31  5214.5 1937.33  5219.8 1938.28  5228.6 1938.27
  5272.6 1937.67  5291.1  1936.8  5322.6 1936.77    5381 1937.72  5552.4 1938.91
#Mann= 3 ,-1 , 0
  4351.1     .05       0  4993.4     .05       0  5001.3     .05       0
Bank Sta=4993.4,5001.3
XS Rating Curve= 0 ,0
Exp/Cntr=0.3,0.1

Type RM Length L Ch R = 1 ,89526   ,329,329,329
BEGIN DESCRIPTION:
Lytle Creek 89915
END DESCRIPTION:
XS GIS Cut Line= 5
      1624592.08      6794937.41      1624688.25      6795198.63
      1624731.81        6795390.      1624761.34      6795599.28
      1625170.32      6795772.68
#Sta/Elev= 30
  4538.2 1938.12  4570.8 1937.31  4602.8 1937.14  4649.3 1935.42  4741.3 1933.46
  4760.5 1933.65  4822.7  1932.9  4827.9  1933.2  4928.7  1932.1  4949.2  1933.1
  4969.8 1932.85    4980  1931.6  4986.3 1926.85  4987.5 1926.35    4993 1926.35
  4994.2 1926.85  5020.9 1932.64  5051.2  1934.5  5068.9 1933.97  5211.2  1933.7
  5357.4 1935.16  5515.8  1935.8  5563.1 1936.65  5568.5 1936.39  5592.2 1937.45
  5597.6 1937.11  5621.3 1937.58  5639.5 1936.77    5645  1937.4  5668.4 1936.21
#Mann= 3 ,-1 , 0
  4538.2     .05       0  4986.3     .05       0  4994.2     .05       0
Bank Sta=4986.3,4994.2
XS Rating Curve= 0 ,0
Exp/Cntr=0.3,0.1

Type RM Length L Ch R = 1 ,89197   ,169,169,169
BEGIN DESCRIPTION:
Lytle Creek 89547.78
END DESCRIPTION:
XS GIS Cut Line= 4
      1624395.83      6794978.53      1624411.02      6795395.18
        1624410.       6795531.4      1624404.48      6796458.33
#Sta/Elev= 30
  4591.8 1935.29  4731.4 1933.79  4741.4 1934.04  4801.4 1932.81  4851.4 1932.24
  4861.4 1932.49  4871.5  1931.9  4881.5  1932.2  4911.5 1931.75  4941.5 1931.91
  4971.5 1930.79  4978.6 1931.44  4983.6 1930.89  4987.6 1927.11  4988.7 1926.61
  4994.3 1926.61  4995.5 1927.11  5001.5 1928.44  5007.6 1930.69  5021.5 1930.07
  5051.5 1932.06  5061.5 1931.28  5091.5 1930.88  5321.6 1929.64  5571.6 1929.05
  5691.6  1928.1  5881.6  1928.4  5921.6 1928.89  5991.6 1932.51  6071.9 1934.28
#Mann= 3 ,-1 , 0
  4591.8     .05       0  4987.6     .05       0  4995.5     .05       0
#XS Ineff= 2 , 0
       0                  5035.8       0 1934.04
Permanent Ineff=
       F       F
Bank Sta=4987.6,4995.5
XS Rating Curve= 0 ,0
Exp/Cntr=0.3,0.1

Type RM Length L Ch R = 1 ,89028   ,697,697,697
BEGIN DESCRIPTION:
Lytle Creek 89363.56
END DESCRIPTION:
XS GIS Cut Line= 5
      1624243.92      6794952.48      1624259.11      6795399.52
      1624264.58      6795801.57      1624299.15      6795898.07
       1624303.7      6796487.56
#Sta/Elev= 30
  4559.5 1933.55  4705.1 1933.07  4935.2 1929.77  4985.3 1930.14  4987.6 1926.32
  4988.7 1925.82    5001 1926.32  5003.5 1929.11  5015.3 1928.88  5045.3 1930.55
  5095.3 1930.31  5105.3 1930.69  5125.3  1930.2  5205.3 1930.09  5235.3 1930.52
  5365.3 1928.89  5375.3 1929.43  5385.3 1928.92  5453.8 1928.21  5479.2 1928.68
  5508.7  1928.1  5571.3 1927.79  5641.3 1927.94  5861.3 1927.26  5891.3 1928.17
  5911.3 1928.25  5981.3 1931.27  6001.3 1931.34  6071.3 1933.38  6100.9  1933.4
#Mann= 3 ,-1 , 0
  4559.5     .05       0  4987.6     .05       0    5001     .05       0
#XS Ineff= 2 , 0
       0                    5091       0  1932.3
Permanent Ineff=
       F       F
Bank Sta=4987.6,5001
XS Rating Curve= 0 ,0
Exp/Cntr=0.3,0.1

Type RM Length L Ch R = 1 ,88331   ,309,309,309
BEGIN DESCRIPTION:
Lytle Creek 88641.42
END DESCRIPTION:
XS GIS Cut Line= 4
      1623805.32      6795581.36      1624153.64      6795739.78
      1624264.81      6795890.07      1624288.72      6796461.68
#Sta/Elev= 30
  4618.6 1929.59    4767 1928.05  4795.6 1928.17  4881.9 1926.81  4887.8 1927.07
  4980.1 1926.63  4991.8 1925.96  4999.3 1924.82  5003.3 1924.82  5004.6 1923.22
  5005.8 1922.72  5011.5 1922.72  5012.7 1923.22  5014.8 1925.22  5023.2 1928.74
  5129.7 1928.49  5150.5 1927.99  5326.2 1927.31  5346.3 1926.88  5356.3 1927.27
  5396.3 1927.26  5446.3  1926.6  5456.4 1927.28  5476.4 1926.77  5526.4 1926.56
  5596.5  1928.6  5626.5 1929.08  5656.5 1930.62  5706.6 1932.09  5760.3 1932.96
#Mann= 3 ,-1 , 0
  4618.6     .05       0  5004.6     .05       0  5012.7     .05       0
#XS Ineff= 2 , 0
       0                  5028.3       0 1930.35
Permanent Ineff=
       F       F
Bank Sta=5004.6,5012.7
XS Rating Curve= 0 ,0
Exp/Cntr=0.3,0.1

Type RM Length L Ch R = 1 ,88022   ,644,644,644
BEGIN DESCRIPTION:
Lytle Creek 88332.5
END DESCRIPTION:
XS GIS Cut Line= 4
      1623691.45      6795732.46      1623908.45      6795895.21
      1624263.83      6796024.92      1624266.64      6796459.75
#Sta/Elev= 30
  4729.7 1931.41  4779.2 1930.86  4793.8 1930.99  4808.4 1931.83  4821.6 1930.85
  4921.6 1928.55  4935.5 1925.63  4950.1 1924.81  4964.7 1923.13  4974.5 1922.84
  4995.1 1922.66  4996.3 1922.16    5002 1922.16  5003.2 1922.66  5018.5 1923.78
  5023.8 1922.74  5029.2 1925.61  5115.4 1927.03  5170.9 1926.85  5242.1 1927.08
  5274.1 1926.58  5422.9 1927.21  5502.3 1926.55  5522.8 1926.98  5532.3 1927.17
  5542.3 1926.55  5592.3 1926.69  5662.3 1928.36  5732.3 1931.01  5814.1 1932.49
#Mann= 7 ,-1 , 0
  4729.7     .05       0  4974.5     .12       0  4995.1     .07       0
  5003.2     .12       0  5170.9     .05       0  5422.9     .12       0
  5522.8     .05       0
#XS Ineff= 2 , 0
       0  4868.3 1929.42  5131.7       0 1929.42
Permanent Ineff=
       F       F
Bank Sta=4995.1,5003.2
XS Rating Curve= 0 ,0
Exp/Cntr=0.3,0.1

Type RM Length L Ch R = 1 ,87378   ,476,476,476
BEGIN DESCRIPTION:
Lytle Creek 87790.86
END DESCRIPTION:
XS GIS Cut Line= 3
      1623443.73      6796084.55      1623636.15      6796478.55
      1623991.01      6796579.83
#Sta/Elev= 30
  4650.4 1926.31  4676.5 1924.75  4743.3 1922.16  4797.4 1922.21    4810 1922.72
  4943.6 1922.36  4954.7 1921.79  4966.2  1919.1  4983.1 1916.97  4988.7 1915.11
  4994.8 1915.09  4996.1 1914.59  5002.3 1914.59  5003.6 1915.09  5021.5 1917.51
  5028.2 1921.34  5043.7 1923.34  5073.2 1923.59  5078.8 1922.07  5090.9 1922.51
  5098.1 1921.84  5104.2 1922.98  5109.4 1922.32  5118.9 1923.03  5170.9 1922.59
  5210.8 1923.52    5216 1922.82  5283.7 1923.61  5288.9 1923.12  5457.9 1925.85
#Mann= 3 ,-1 , 0
  4650.4     .05       0  4994.8     .05       0  5003.6     .05       0
Bank Sta=4994.8,5003.6
XS Rating Curve= 0 ,0
Exp/Cntr=0.3,0.1

Type RM Length L Ch R = 1 ,86902   ,255,255,255
BEGIN DESCRIPTION:
Lytle Creek 87176.58
END DESCRIPTION:
XS GIS Cut Line= 3
      1623401.56      6796134.37      1623167.21      6796590.06
      1623114.26       6796711.5
#Sta/Elev= 30
  4512.1  1924.3  4518.7 1924.96  4535.2 1923.78  4585.2 1923.12  4617.4 1922.26
  4623.9 1921.47  4629.5 1921.97  4639.9 1921.68  4646.1 1921.04  4795.7 1920.07
  4840.1  1920.3  4862.3 1919.77  4884.4 1920.63  4943.5 1920.52  4956.6 1920.13
  4973.1  1915.5  4978.8 1915.71  4988.5 1913.99  5006.6 1913.51  5007.9 1913.01
  5014.1 1913.01  5015.4 1913.51  5017.5 1914.09  5024.5 1914.34    5046 1917.15
    5055 1919.85    5064 1921.39  5069.5  1921.3  5087.4 1919.55    5157 1918.77
#Mann= 3 ,-1 , 0
  4512.1     .05       0  5006.6     .05       0  5015.4     .05       0
Bank Sta=5006.6,5015.4
XS Rating Curve= 0 ,0
Exp/Cntr=0.3,0.1

Type RM Length L Ch R = 1 ,86647   ,712,712,712
BEGIN DESCRIPTION:
Lytle Creek 86919.68
END DESCRIPTION:
XS GIS Cut Line= 4
      1623109.93      6796103.05      1622940.65       6796493.7
      1622823.46      6796755.51      1622836.59      6797017.49
#Sta/Elev= 30
  4544.4 1929.08  4596.7 1929.02  4713.3 1927.17  4811.4 1926.51  4842.3 1924.89
  4871.2 1924.28  4909.4 1922.37  4931.2 1920.03  4941.7 1917.84  4947.1 1917.31
    4953 1914.63  4969.8 1913.21  4993.8 1912.69  4994.8 1912.19  4996.1 1911.69
  5002.4 1911.69  5003.6 1912.19  5022.4 1916.01  5029.6 1918.13  5045.6 1918.72
  5097.5 1918.62  5115.2 1918.03  5138.4 1919.25  5161.1 1918.12  5204.9 1917.14
  5386.1 1916.41  5419.7 1916.61  5439.7 1917.65  5479.8 1916.54  5519.3 1918.09
#Mann= 3 ,-1 , 0
  4544.4     .05       0  4994.8     .03       0  5003.6     .05       0
Bank Sta=4994.8,5003.6
XS Rating Curve= 0 ,0
Exp/Cntr=0.3,0.1

Type RM Length L Ch R = 1 ,85935   ,525,525,525
BEGIN DESCRIPTION:
Lytle Creek 86174.52
END DESCRIPTION:
XS GIS Cut Line= 4
      1622294.38      6796181.76      1622304.79      6796747.69
      1622303.09      6796815.98       1622733.2      6797162.07
#Sta/Elev= 30
  4443.1 1919.45  4509.4 1920.24  4599.4 1919.86  4609.4 1920.18  4619.4 1921.95
  4629.4 1923.09  4679.4 1923.01  4709.4  1923.7  4819.4  1924.4  4859.4  1923.8
  4919.4 1922.41  4939.4 1921.12  4949.4 1918.41  4989.4 1910.63  5002.3 1909.79
  5003.6 1909.29  5009.9 1909.29  5011.2 1909.79  5039.4 1914.63  5049.5 1915.35
  5075.9 1913.64  5087.5  1913.5  5093.9 1912.94  5122.7 1912.91  5157.9 1913.38
  5272.4 1913.36  5372.2 1913.92    5585 1913.96  5620.2 1914.29  5629.5 1915.53
#Mann= 3 ,-1 , 0
  4443.1     .05       0  5002.3     .05       0  5011.2     .05       0
Bank Sta=5002.3,5011.2
XS Rating Curve= 0 ,0
Exp/Cntr=0.3,0.1

Type RM Length L Ch R = 1 ,85410   ,239,239,239
BEGIN DESCRIPTION:
Lytle Creek 85633.84
END DESCRIPTION:
XS GIS Cut Line= 4
      1621777.02      6796167.81      1621794.38      6796744.22
      1621808.59      6797090.17      1622248.12      6797164.64
#Sta/Elev= 30
  4414.9 1914.93  4495.1 1913.84  4535.1 1913.75  4575.2 1912.89  4615.2 1913.55
  4695.2 1912.24  4745.2 1912.15  4843.2 1910.62  4875.3 1910.51  4975.3 1911.55
    4991 1908.45    4996 1908.45  5000.9 1905.83  5002.2 1905.33  5008.5 1905.33
  5009.8 1905.83  5015.4 1910.96  5025.4 1911.62  5045.4  1911.8  5065.4 1910.86
  5085.4 1910.49  5175.5 1910.76  5364.6 1909.69  5435.6 1910.28  5472.8 1911.04
  5477.8 1910.83  5496.4 1911.14  5567.4 1910.99  5653.9 1911.64  5783.6 1911.88
#Mann= 3 ,-1 , 0
  4414.9     .05       0  5000.9     .05       0  5009.8     .05       0
Bank Sta=5000.9,5009.8
XS Rating Curve= 0 ,0
Exp/Cntr=0.3,0.1

Type RM Length L Ch R = 1 ,85171   ,321,321,321
BEGIN DESCRIPTION:
Lytle Creek 85399.18
END DESCRIPTION:
XS GIS Cut Line= 4
       1621554.8      6796133.14      1621575.63      6796695.61
      1621570.54      6797262.98      1621638.62      6797397.03
#Sta/Elev= 30
  4444.8 1916.15  4499.7 1916.17  4529.7 1914.83  4579.8 1914.14  4669.8 1913.99
  4679.8 1913.12  4709.8 1912.26  4739.9 1911.96  4799.9 1910.27  4809.9 1910.59
  4855.3 1909.12    4910 1908.37    4970 1909.41    4980 1908.78  4985.6 1904.23
  4986.9 1903.73  4993.2 1903.73  4994.5 1904.23  5006.4 1908.51  5011.4 1908.51
    5020 1910.79    5030 1909.63    5060 1909.53    5090 1908.42  5170.1 1907.59
  5380.1 1908.06  5580.7 1907.46  5657.9 1907.66  5685.8 1908.26  5725.4 1908.42
#Mann= 3 ,-1 , 0
  4444.8     .05       0  4985.6     .03       0  4994.5     .05       0
Bank Sta=4985.6,4994.5
XS Rating Curve= 0 ,0
Exp/Cntr=0.3,0.1

Type RM Length L Ch R = 1 ,84850   ,253,253,253
BEGIN DESCRIPTION:
Mapping XS dbb66543
END DESCRIPTION:
XS GIS Cut Line= 4
       1621177.2        6796135.      1621218.88      6796437.13
      1621319.57      6797076.02      1621639.07      6797440.29
#Sta/Elev= 30
  4416.8 1916.35    4585  1915.9  4601.5 1916.27  4631.8 1915.27  4641.9 1915.51
  4651.9 1916.38  4672.2 1915.48  4728.4 1915.06  4839.2  1913.2  4884.6 1912.35
  4923.3 1910.85  4975.8 1907.78  4983.4 1905.82  4988.4 1905.87  4991.5 1904.88
  4992.8 1904.38  4999.2 1904.38  5000.5 1904.88  5006.1 1905.54  5016.3 1907.64
  5026.4 1907.81  5097.2 1906.44  5243.4 1906.79    5367 1905.26  5451.4  1906.9
  5657.3 1906.54    5792 1907.16  5820.5  1907.4  5841.4 1908.15  5853.1 1907.98
#Mann= 5 ,-1 , 0
  4416.8     .05       0  4839.2     .12       0  4923.3     .05       0
  4991.5     .05       0  5000.5     .05       0
Bank Sta=4991.5,5000.5
XS Rating Curve= 0 ,0
Exp/Cntr=0.3,0.1

Type RM Length L Ch R = 1 ,84597   ,955,955,955
BEGIN DESCRIPTION:
Lytle Creek 84881.32
END DESCRIPTION:
XS GIS Cut Line= 4
      1620922.84      6796414.33      1621058.27      6796692.14
      1621194.35      6797000.21      1621643.34       6797496.5
#Sta/Elev= 30
  4679.4 1912.28  4855.7 1914.74  4928.9  1914.7  4951.4 1914.18  4961.6 1913.42
  4968.4 1911.74  4973.9 1908.58  4983.4 1905.33  4988.5 1905.33  4991.1 1903.97
  4996.5 1902.71  5001.3 1902.24  5002.6 1901.74    5009 1901.74  5010.3 1902.24
  5019.8 1905.37  5037.7 1906.19  5071.9 1905.91  5113.1 1904.76  5292.6 1905.38
  5331.3 1904.81  5394.9 1905.23    5480 1904.79  5592.9 1906.71  5926.1 1906.63
  5968.7 1907.17  5975.5 1907.71  5989.7  1907.8  5992.2 1908.43  5994.5 1908.43
#Mann= 3 ,-1 , 0
  4679.4     .05       0  5001.3     .05       0  5010.3     .05       0
Bank Sta=5001.3,5010.3
XS Rating Curve= 0 ,0
Exp/Cntr=0.3,0.1

Type RM Length L Ch R = 1 ,83642   ,431,431,431
BEGIN DESCRIPTION:
Mapping XS f6a1cfaa
END DESCRIPTION:
XS GIS Cut Line= 4
      1620816.09      6796423.29      1620740.58      6796928.45
      1620925.48      6797425.85       1621296.8      6797368.84
#Sta/Elev= 30
  4257.2 1910.07  4564.6 1908.59    4626 1907.81  4633.8 1907.49  4638.9 1906.42
  4696.7 1905.71  4747.3 1904.38  4770.4 1905.17  4794.6 1903.99    4850 1903.12
  4971.4 1902.38  4980.9  1899.6  4991.1 1898.08  4996.4 1898.38  5008.3 1897.57
  5009.6 1897.07  5016.1 1897.07  5017.4 1897.57  5021.4 1899.51  5026.7 1898.37
  5044.9 1901.03  5082.1 1901.56  5098.2 1901.28  5119.6 1901.83  5162.2  1901.1
  5258.9 1902.43  5452.1 1902.44  5561.2 1903.66  5601.7 1904.66  5674.3 1904.54
#Mann= 3 ,-1 , 0
  4257.2     .05       0  5008.3     .05       0  5017.4     .05       0
Bank Sta=5008.3,5017.4
XS Rating Curve= 0 ,0
Exp/Cntr=0.3,0.1
