HEC-RAS study Lytle Creek.prj: Lytle Creek Base Level Engineering

--- Lytle Creek.g02 (geometry) --- (continued)

Type RM Length L Ch R = 1 ,60250   ,298,298,298
BEGIN DESCRIPTION:
Lytle Creek 61296.893
END DESCRIPTION:
XS GIS Cut Line= 3
      1610937.47      6807247.22      1611354.85      6807312.79
      1612315.92      6807240.26
#Sta/Elev= 30
  4577.5 1813.19  4726.8 1814.09  4777.5 1813.24  4797.7    1811  4817.9 1811.91
  4838.2 1810.77  4873.1 1810.78  4888.8 1809.42    4909 1808.69  4929.3 1806.16
  4940.7  1805.8  4952.7 1801.11  4954.2 1800.61  4965.2 1800.61  4966.7 1801.11
    4990 1801.89  5002.6 1801.38  5020.2  1802.4  5040.3 1806.83  5060.3 1808.96
  5132.8 1809.79  5140.5 1810.76  5220.8    1812  5270.9 1811.26  5491.5 1812.25
  5532.7 1811.39    5652 1810.86  5772.3 1813.58  5842.5 1816.05  5963.8 1817.53
#Mann= 3 ,-1 , 0
  4577.5     .05       0  4952.7     .05       0  4966.7     .05       0
Bank Sta=4952.7,4966.7
XS Rating Curve= 0 ,0
Exp/Cntr=0.3,0.1

Type RM Length L Ch R = 1 ,59952   ,189,189,189
BEGIN DESCRIPTION:
Lytle Creek 60583.97
END DESCRIPTION:
XS GIS Cut Line= 5
      1611165.87      6807304.29      1611235.56       6807436.7
      1611235.56      6807590.65      1611262.68      6807928.99
      1611266.12      6808710.18
#Sta/Elev= 30
    4724 1811.44  4771.8  1811.1  4777.4 1810.13  4793.8 1809.84  4829.9 1809.75
  4843.5 1808.79  4884.9 1808.26  4954.9 1804.92  4964.9  1805.1  4994.9 1800.38
  5007.9 1799.44  5009.4 1798.94  5020.4 1798.94  5021.9 1799.44  5023.8 1800.63
  5027.6 1800.63    5035 1804.51    5055 1807.03  5081.6 1809.31  5145.3  1807.6
  5215.5 1807.15  5337.2 1808.94    5556 1807.72    5576 1807.12    5596 1808.01
    5676 1807.01    5796  1807.6    5996  1810.8    6086 1810.46  6148.2 1812.08
#Mann= 3 ,-1 , 0
    4724     .05       0  5007.9     .03       0  5021.9     .05       0
Bank Sta=5007.9,5021.9
XS Rating Curve= 0 ,0
Exp/Cntr=0.3,0.1

Type RM Length L Ch R = 1 ,59763   ,280,280,280
BEGIN DESCRIPTION:
Lytle Creek 60407.03
END DESCRIPTION:
XS GIS Cut Line= 4
      1611072.37      6807417.06      1611100.14      6807694.82
      1611104.59      6808004.37       1611190.3      6808409.27
#Sta/Elev= 30
  4721.8 1811.75  4762.9 1810.96    4783 1811.15  4798.3 1809.14  4883.5 1807.67
  4893.6 1807.14  4903.8 1805.21  4923.7 1803.83  4943.8 1803.34  4953.9 1802.45
  4963.9 1800.77  4987.1 1799.16  4988.6 1798.66  4999.6 1798.66  5001.1 1799.16
  5014.1 1800.21  5034.1  1803.8  5044.1 1804.43  5054.1 1803.61  5094.1 1803.78
  5144.1 1807.09  5254.2 1807.33  5314.9 1806.76  5432.5 1807.95  5457.3 1807.31
  5467.6 1807.71  5626.2 1806.93  5631.3  1808.1  5720.5 1809.96  5724.4 1809.48
#Mann= 3 ,-1 , 0
  4721.8     .05       0  4987.1     .03       0  5001.1     .05       0
Bank Sta=4987.1,5001.1
XS Rating Curve= 0 ,0
Exp/Cntr=0.3,0.1

Type RM Length L Ch R = 1 ,59483   ,280,280,280
BEGIN DESCRIPTION:
Lytle Creek 60136.79
END DESCRIPTION:
XS GIS Cut Line= 5
       1610268.7      6807202.33      1610738.38      6807688.48
      1610940.42      6807903.15      1611049.39      6808156.85
      1611185.41      6808436.77
#Sta/Elev= 30
  4010.7 1815.24  4089.8 1815.26  4252.6 1813.31  4295.1 1813.81  4365.8 1812.72
  4401.1 1813.28    4408 1813.17  4415.2 1811.68  4443.5 1810.81  4521.2    1812
  4570.8 1809.38  4669.9 1807.29  4832.6 1807.24  4875.1 1808.65  4931.7 1805.75
    4960 1802.18  4981.1 1797.79  4997.4  1797.2  4998.9  1796.7  5011.4  1797.2
  5019.4 1800.69    5028 1802.07  5062.9 1803.91  5080.5 1803.94  5117.3 1807.08
  5156.6 1807.83    5414 1806.31  5503.5 1807.73  5509.8 1808.88  5568.8 1810.42
#Mann= 3 ,-1 , 0
  4010.7     .05       0  4997.4     .05       0  5011.4     .05       0
Bank Sta=4997.4,5011.4
XS Rating Curve= 0 ,0
Exp/Cntr=0.3,0.1

Type RM Length L Ch R = 1 ,59203   ,280,280,280
BEGIN DESCRIPTION:
Lytle Creek 59825.13
END DESCRIPTION:
XS GIS Cut Line= 5
      1610187.99      6807244.02      1610644.12      6808009.17
      1610807.52      6808142.53      1610962.51      6808249.09
      1611178.86      6808464.07
#Sta/Elev= 30
  3878.7 1813.54  4024.1 1811.47  4076.7 1809.63  4135.1 1809.11  4140.9 1810.48
  4156.5 1810.88  4172.1 1809.06  4251.9 1807.78  4740.5 1806.36  4811.5 1807.83
  4840.2 1807.08  4875.4 1807.72  4897.7 1806.78  4918.5  1804.3    4968 1802.06
  4989.5 1797.24  5005.1 1796.54  5006.6 1796.04  5019.1 1796.54  5025.9 1799.75
  5033.1 1800.97  5039.1  1804.1    5048 1804.56    5054 1806.12  5155.5 1806.76
  5268.5 1805.97    5417 1810.21  5445.3 1810.35  5452.3 1809.41  5473.5 1810.52
#Mann= 3 ,-1 , 0
  3878.7     .05       0  5005.1     .05       0  5019.1     .05       0
Bank Sta=5005.1,5019.1
XS Rating Curve= 0 ,0
Exp/Cntr=0.3,0.1

Type RM Length L Ch R = 1 ,58923   ,286,286,286
BEGIN DESCRIPTION:
Lytle Creek 59569.64
END DESCRIPTION:
XS GIS Cut Line= 6
      1609689.42      6808022.75      1609997.74      6808257.34
      1610456.22      6808267.46      1610621.41      6808319.12
      1610867.94       6808359.6      1611177.54       6808488.8
#Sta/Elev= 30
  3981.5 1807.79  4352.9 1805.01  4456.2 1805.95  4566.2 1804.91  4586.2 1804.16
  4623.3 1799.67  4659.3 1799.15  4666.3 1797.48  4669.3  1795.1  4670.8  1794.6
  4683.3  1795.1  4686.3 1797.75  4696.3 1801.17  4716.3 1804.29  4811.9 1805.42
  4868.1 1806.17  4889.1 1803.44  4908.9 1805.39  4914.2 1801.57  4941.4 1806.24
  4946.6 1802.09  4962.4    1803  4993.9 1797.41  5004.9 1797.42  5044.8 1802.78
  5083.9 1804.45    5159 1806.04  5332.8  1805.5  5468.2 1809.33  5585.9 1810.49
#Mann= 7 ,-1 , 0
  3981.5     .05       0  4659.3     .12       0  4669.3     .05       0
  4683.3     .12       0  4811.9     .05       0  5083.9     .12       0
    5159     .05       0
Bank Sta=4669.3,4683.3
XS Rating Curve= 0 ,0
Exp/Cntr=0.3,0.1

Type RM Length L Ch R = 1 ,58637   ,455,455,455
BEGIN DESCRIPTION:
Lytle Creek 59281.01
END DESCRIPTION:
XS GIS Cut Line= 5
      1609649.09      6808099.36      1610554.23      6808586.85
      1610623.58      6808560.01      1610895.12      6808489.41
      1611185.37      6808517.46
#Sta/Elev= 30
  3881.8 1807.88  4230.9 1805.06  4342.8 1805.89    4411 1804.45  4422.4 1801.18
  4438.6  1799.9  4504.3 1799.84  4506.3 1792.99  4507.8 1792.49  4520.3 1792.99
  4520.5 1799.89    4570 1794.49  4586.2 1798.29  4592.7 1802.74  4602.4 1805.29
  4624.4 1804.03  4777.7 1804.26  4948.2 1806.57  4973.5 1800.23    4996 1795.26
  5006.4 1794.64    5017 1799.24  5037.4 1801.62    5120 1800.69    5174 1802.95
  5206.2 1801.23  5214.5 1800.93  5249.9 1804.97  5345.1 1807.89  5556.4 1811.29
#Mann= 5 ,-1 , 0
  3881.8     .05       0  4506.3     .07       0  4520.3     .05       0
  4973.5     .12       0  5206.2     .05       0
Bank Sta=4506.3,4520.3
XS Rating Curve= 0 ,0
Exp/Cntr=0.3,0.1

Type RM Length L Ch R = 1 ,58182   ,529,529,529
BEGIN DESCRIPTION:
Lytle Creek 58794.3
END DESCRIPTION:
XS GIS Cut Line= 5
      1609705.92      6808185.31       1610657.4      6808722.42
      1610781.74      6808827.36      1610905.26      6808859.16
      1611129.25      6808925.58
#Sta/Elev= 30
  3617.7 1806.32  3994.7 1805.95  4081.3 1799.06  4140.5  1799.9  4142.1 1793.05
  4143.6 1792.55  4156.2 1793.05  4156.4 1799.64  4199.7 1798.76  4205.5 1795.61
  4213.8 1794.22  4227.1 1801.55  4236.7 1805.09  4243.1  1805.3  4397.5 1803.75
  4544.9  1805.2  4741.1 1804.55  4776.2 1805.83  4819.1 1803.11  4878.8 1802.26
    4959 1799.35  4975.2 1796.67    5003  1794.9  5009.8 1800.23    5015 1798.26
  5021.2 1804.34  5031.6 1807.17  5043.5 1807.66  5186.4 1807.69  5234.2 1809.35
#Mann= 5 ,-1 , 0
  3617.7     .05       0  4142.1     .07       0  4156.2     .05       0
  4878.8     .12       0  5043.5     .05       0
Bank Sta=4142.1,4156.2
XS Rating Curve= 0 ,0
Exp/Cntr=0.3,0.1

Type RM Length L Ch R = 1 ,57653   ,425,425,425
BEGIN DESCRIPTION:
Lytle Creek 59575.975
END DESCRIPTION:
XS GIS Cut Line= 5
      1609691.65      6808227.01      1610319.43      6808639.07
      1610551.05      6808844.69      1610604.66      6809064.34
      1610958.41      6809261.43
#Sta/Elev= 30
  3856.4  1806.1  4228.5 1804.79  4264.7  1802.3  4291.7 1798.78  4364.1 1799.33
  4373.2 1797.22  4379.2 1793.87  4415.3 1799.24  4430.4 1803.75  4458.5 1805.07
  4502.8 1803.55  4674.2 1803.71  4780.4 1802.34  4941.3 1804.45  4961.6 1805.63
  4971.9 1803.69  4982.2 1798.36  4990.2  1792.4  4991.7  1791.9  5004.4  1792.4
  5023.4 1797.37  5085.8 1797.51  5109.1 1800.56  5176.8 1804.81  5224.2 1805.84
  5256.1 1806.69  5372.5 1807.41  5404.3 1808.73  5431.7 1807.49  5548.1 1807.83
#Mann= 7 ,-1 , 0
  3856.4     .05       0  4941.3     .12       0  4990.2     .07       0
  5004.4     .12       0  5109.1     .05       0  5224.2     .12       0
  5256.1     .05       0
Bank Sta=4990.2,5004.4
XS Rating Curve= 0 ,0
Exp/Cntr=0.3,0.1

Type RM Length L Ch R = 1 ,57228   ,459,459,459
BEGIN DESCRIPTION:
Lytle Creek 57862.05
END DESCRIPTION:
XS GIS Cut Line= 3
      1609411.92      6808436.71      1610251.88      6809147.27
      1610788.35      6809220.19
#Sta/Elev= 30
  3914.5 1806.96  3924.7 1806.07  3945.5  1805.8  4300.4  1803.8    4797 1802.28
  4839.9 1802.51  4868.4 1803.86    4897 1803.04  4953.3 1803.31  4967.3 1802.83
    4975 1799.11  4981.6 1800.19  4989.3 1793.22  4995.9 1794.91  5005.5 1790.71
    5007 1790.21  5021.5 1790.71  5027.9 1795.07    5038 1795.95  5055.2 1795.11
  5068.3 1796.82  5088.5 1797.46  5132.7 1797.45  5199.5 1800.45  5229.8 1799.98
  5300.4 1804.05  5320.6  1804.1  5391.2 1806.47  5432.6 1807.36  5556.1 1808.02
#Mann= 3 ,-1 , 0
  3914.5     .05       0  5005.5     .05       0  5021.5     .05       0
Bank Sta=5005.5,5021.5
XS Rating Curve= 0 ,0
Exp/Cntr=0.3,0.1

Type RM Length L Ch R = 1 ,56769   ,381,381,381
BEGIN DESCRIPTION:
Lytle Creek 57486.78
END DESCRIPTION:
XS GIS Cut Line= 5
      1609318.17      6808457.54      1610113.45      6809201.79
       1610202.4      6809444.15      1610318.99      6809684.41
      1610520.03      6809768.11
#Sta/Elev= 30
  3636.5 1805.93  4129.8 1803.06  4646.1 1801.69  4726.3 1802.42  4771.7 1801.44
  4785.6  1802.2  4811.9  1801.7  4832.7 1799.86  4849.5 1795.04  4857.8  1794.6
  4893.6 1794.85  4913.4 1797.25    4937 1795.87    4956 1796.57  4974.5 1795.73
  4979.8 1794.41  4983.3 1791.94  4988.8 1791.94  4995.1 1788.45  4996.6 1787.95
  5011.1 1788.45  5020.1 1795.26  5032.6 1800.59  5042.6 1803.24  5087.8 1801.91
    5161 1801.75  5321.2 1804.55  5326.6 1803.73  5355.8 1804.94  5468.7 1805.39
#Mann= 6 ,-1 , 0
  3636.5     .05       0  4726.3     .12       0  4811.9     .05       0
    4937     .12       0  4995.1     .07       0  5011.1     .05       0
Bank Sta=4995.1,5011.1
XS Rating Curve= 0 ,0
Exp/Cntr=0.3,0.1

Type RM Length L Ch R = 1 ,56388   ,350,350,350
BEGIN DESCRIPTION:
Lytle Creek 57107.41
END DESCRIPTION:
XS GIS Cut Line= 5
      1609394.43      6808601.22      1609841.84      6809216.51
      1609869.06      6809389.46      1609923.19      6809594.01
      1610233.94        6809737.
#Sta/Elev= 30
  4105.6 1804.99  4389.7 1802.87  4839.2 1801.96  4888.1 1803.09  4916.1 1802.13
  4921.2 1800.97  4938.7 1799.58    4959 1796.33  4978.6 1790.23  4983.7 1793.57
  4989.3 1789.84  4991.5  1787.1    4993  1786.6  5007.5  1787.1  5009.6 1789.12
  5019.7 1790.66  5057.1 1794.17    5071 1794.89  5080.2 1796.43  5085.3 1795.93
  5112.3 1799.65  5131.9 1800.26  5220.6  1801.8  5256.8 1801.45    5266 1800.69
  5324.5 1800.57  5530.2 1802.75  5552.2 1802.26  5565.2 1803.08  5595.1 1803.26
#Mann= 7 ,-1 , 0
  4105.6     .05       0  4839.2     .12       0  4991.5     .07       0
  5007.5     .12       0  5057.1     .05       0  5131.9     .12       0
  5220.6     .05       0
Bank Sta=4991.5,5007.5
XS Rating Curve= 0 ,0
Exp/Cntr=0.3,0.1

Type RM Length L Ch R = 1 ,56038   ,273,273,273
BEGIN DESCRIPTION:
Mapping XS 555dad79
END DESCRIPTION:
XS GIS Cut Line= 5
      1609351.83      6808569.23      1609401.84      6809291.85
      1609833.83      6809520.07       1609921.3      6809602.31
      1610219.82      6809739.93
#Sta/Elev= 30
  4047.2 1805.17    4477 1802.08  4567.2 1802.76  4596.2 1801.56  4767.1 1800.51
  4956.1 1801.14  4964.2 1799.21  4969.9 1801.17  4978.2 1786.52  4979.7 1786.02
  4994.2 1786.52  5001.3 1787.16  5008.2 1789.69  5013.9 1788.18  5030.3  1791.6
  5035.9 1789.92  5052.3 1794.38  5060.5 1794.96  5112.7 1795.47  5134.7 1794.05
  5140.3 1792.81  5156.7 1794.75  5162.3 1796.62  5216.2 1794.29  5222.7 1798.27
  5228.4 1797.45  5238.8 1799.39  5359.5 1801.13  5472.1 1800.69  5708.9 1803.08
#Mann= 5 ,-1 , 0
  4047.2     .05       0  4978.2     .05       0  4994.2     .05       0
  5060.5     .12       0  5359.5     .05       0
Bank Sta=4978.2,4994.2
XS Rating Curve= 0 ,0
Exp/Cntr=0.3,0.1

Type RM Length L Ch R = 1 ,55765   ,171,171,171
BEGIN DESCRIPTION:
Lytle Creek 56486.22
END DESCRIPTION:
XS GIS Cut Line= 5
       1609336.8      6809055.48      1609442.13      6809658.26
      1609652.92      6809660.29       1609906.1      6809666.05
      1610187.89      6809736.79
#Sta/Elev= 30
  4171.3  1802.4  4303.4 1800.95  4691.6 1799.48  4846.1 1799.62  4946.1 1801.27
  4956.1 1799.52  4976.1 1791.89  4984.6 1785.98  4986.1 1785.48  5000.6 1785.98
  5006.1  1786.2  5016.1 1791.01  5026.1 1793.78  5056.1 1795.61  5066.1 1794.62
    5085 1794.39  5096.1 1795.69  5106.1 1797.93  5112.2 1798.16  5156.1 1796.74
  5196.2 1797.26  5206.2 1798.45  5220.8 1798.78  5256.4 1801.16  5287.4 1800.33
  5402.5 1802.02  5438.5 1802.08  5452.3 1801.38  5484.8 1802.54  5537.8 1802.92
#Mann= 5 ,-1 , 0
  4171.3     .05       0  4984.6     .05       0  5000.6     .05       0
    5085     .12       0  5220.8     .05       0
Bank Sta=4984.6,5000.6
XS Rating Curve= 0 ,0
Exp/Cntr=0.3,0.1

Type RM Length L Ch R = 1 ,55594   ,722,722,722
BEGIN DESCRIPTION:
Lytle Creek 56301.97
END DESCRIPTION:
XS GIS Cut Line= 5
      1609315.97      6809071.02      1609426.48      6809653.98
      1609502.01      6809839.51      1609736.25      6809819.15
      1610227.36      6809817.01
#Sta/Elev= 30
  3990.8 1802.78  4007.7 1801.81  4048.8 1801.28  4252.4 1800.22  4498.7 1799.37
  4610.1 1799.56  4671.3 1800.92  4695.3 1800.18  4807.5 1799.41  4856.2  1797.3
  4861.2 1797.58  4968.1 1794.04  4974.1 1790.15  4990.3 1786.22  4991.8 1785.72
  5004.8 1785.72  5006.3 1786.22  5008.3 1786.31  5015.6 1788.88  5019.6 1789.16
  5028.3 1792.59  5038.3 1793.48  5114.6 1794.74  5138.3 1796.91  5158.3 1800.07
  5178.3  1799.5  5198.3 1801.14  5228.3 1800.44  5298.3 1800.62  5510.7 1802.75
#Mann= 5 ,-1 , 0
  3990.8     .05       0  4990.3     .03       0  5006.3     .05       0
  5015.6    .075       0  5114.6     .05       0
Bank Sta=4990.3,5006.3
XS Rating Curve= 0 ,0
Exp/Cntr=0.3,0.1

Type RM Length L Ch R = 1 ,54872   ,646,646,646
BEGIN DESCRIPTION:
Lytle Creek 55798.38
END DESCRIPTION:
XS GIS Cut Line= 4
      1609269.83      6810369.96      1609583.17       6810399.3
      1609975.54      6810382.47      1610709.79      6809975.97
#Sta/Elev= 30
  4807.3 1797.82  4947.6 1797.75  4963.1 1794.54  4973.2 1788.43  4983.2 1785.53
  4995.3 1785.17  4996.8 1784.67  5009.8 1784.67  5011.3 1785.17  5013.4 1787.49
  5023.4 1790.23  5056.5 1792.59  5083.7 1793.46  5113.8 1798.52  5120.4 1798.99
  5125.4 1798.99  5133.9 1795.79  5143.9 1795.67  5163.9 1795.95  5173.9 1796.97
  5183.9 1796.37  5203.9 1796.38    5269 1798.22  5354.1  1799.4  5384.1 1798.99
  5798.4 1799.89    5937 1801.58  6062.8 1801.63  6200.3 1803.22    6354 1803.86
#Mann= 3 ,-1 , 0
  4807.3     .05       0  4995.3     .03       0  5011.3     .05       0
Bank Sta=4995.3,5011.3
XS Rating Curve= 0 ,0
Exp/Cntr=0.3,0.1

Type RM Length L Ch R = 1 ,54226   ,300,300,300
BEGIN DESCRIPTION:
Lytle Creek 55595.381
END DESCRIPTION:
XS GIS Cut Line= 5
       1608870.7      6810524.27      1609654.48      6810972.78
      1609720.92      6810982.35      1609900.61      6810472.27
      1610103.31      6810341.85
#Sta/Elev= 30
  4106.4 1797.17  4228.5 1796.25  4318.7 1796.53  4595.3 1795.21  4668.9 1795.32
  4765.3  1790.8  4802.6 1790.04  4830.1 1789.93  4926.5 1791.33  4969.7 1790.88
  4975.5  1787.2  4991.2 1785.14  4998.5 1785.22  4998.9 1784.61  5000.4 1784.11
  5013.4 1784.11  5014.9 1784.61  5030.2 1788.31  5040.3 1793.69  5060.5 1797.43
  5081.5 1796.84  5229.6 1798.21  5342.8  1798.3  5435.7 1797.63  5568.9 1798.91
  5637.5 1798.89    5682 1799.43  5797.9 1799.15  5840.2 1799.74  5858.4 1799.54
#Mann= 3 ,-1 , 0
  4106.4     .05       0  4998.9    .035       0  5014.9     .05       0
Bank Sta=4998.9,5014.9
XS Rating Curve= 0 ,0
Exp/Cntr=0.3,0.1

Type RM Length L Ch R = 1 ,53926   ,762,762,762
BEGIN DESCRIPTION:
Lytle Creek 54428.227
END DESCRIPTION:
XS GIS Cut Line= 4
      1608783.04      6810569.69      1609001.97      6810980.83
      1609511.97      6811231.46      1610674.64      6811780.87
#Sta/Elev= 30
  3973.2 1796.77  4240.4 1794.91  4670.7 1794.83  4687.5 1793.17  4693.2  1791.8
  4715.7 1790.56  4760.6 1791.34  4850.6  1790.5  4910.4 1791.74    4946 1790.51
  4991.5 1784.41    4993 1783.91  5007.5 1784.41  5030.7 1789.82  5043.8 1794.76
  5165.5 1796.88  5241.1 1797.21  5263.9 1795.61  5298.2 1790.74  5309.2 1791.87
    5315  1793.5  5331.4 1794.25  5383.2 1794.95  5457.1 1794.53  5525.4 1796.11
  5900.6 1795.63  5983.9 1796.22  6171.9 1800.09  6224.8 1802.48  6293.2 1804.12
#Mann= 3 ,-1 , 0
  3973.2     .05       0  4991.5    .035       0  5007.5     .05       0
Bank Sta=4991.5,5007.5
XS Rating Curve= 0 ,0
Exp/Cntr=0.3,0.1

Type RM Length L Ch R = 1 ,53164   ,390,390,390
BEGIN DESCRIPTION:
Lytle Creek 53829.901
END DESCRIPTION:
XS GIS Cut Line= 4
      1608656.59      6810764.74      1608607.73      6811434.22
      1608965.91      6811626.96      1610704.98      6812687.99
#Sta/Elev= 30
    3922 1795.05    4186 1793.55  4910.5  1792.3  4942.2 1791.77  4976.3  1784.8
  5000.2 1783.22  5001.7 1782.72  5016.2 1783.22  5035.4 1788.38  5108.9  1792.1
  5298.6 1792.46  5393.5 1793.83  5451.6 1789.18  5552.3 1789.25  5573.6 1790.75
  5794.2  1790.1  5821.4 1793.36  5830.7 1793.18  5842.7 1790.33  5858.2 1789.55
  5873.6 1786.85  5894.9 1787.28  5924.4 1793.63  5947.2 1794.93  5974.3 1798.43
  6047.9 1800.53  6258.9 1800.04  6417.7 1802.91  6475.8 1802.25  7037.2 1808.31
#Mann= 3 ,-1 , 0
    3922     .05       0  5000.2    .035       0  5016.2     .05       0
Bank Sta=5000.2,5016.2
XS Rating Curve= 0 ,0
Exp/Cntr=0.3,0.1

Type RM Length L Ch R = 1 ,52774   ,362,362,362
BEGIN DESCRIPTION:
Lytle Creek 53266.654
END DESCRIPTION:
XS GIS Cut Line= 4
      1608637.64      6810713.04      1608531.31      6811727.05
      1608757.24      6811943.93      1610130.15      6813115.98
#Sta/Elev= 30
    3645  1795.3  4001.4 1793.17  4487.5 1794.17  4809.2 1791.03  4936.5 1792.05
  4950.7 1790.78  4957.9 1788.03  4972.1 1785.46  4977.1 1783.02  4999.4 1780.88
  5000.9 1780.38  5015.4 1780.88  5021.7 1786.46  5042.5 1786.31  5078.8 1788.39
  5099.6  1786.8  5113.9 1789.86  5134.7 1792.02  5376.3 1791.13  5454.2 1787.53
  5489.4 1787.17  5617.8 1790.03  5695.8 1789.15  5730.9 1790.76  5751.8 1786.07
  5773.7 1785.48  5802.3 1793.19  5829.7 1795.64  5958.2 1797.69  6782.9 1803.25
#Mann= 3 ,-1 , 0
    3645     .05       0  4999.4    .035       0  5015.4     .05       0
Bank Sta=4999.4,5015.4
XS Rating Curve= 0 ,0
Exp/Cntr=0.3,0.1

Type RM Length L Ch R = 1 ,52412   ,1015,1015,1015
BEGIN DESCRIPTION:
Lytle Creek 52677.451
END DESCRIPTION:
XS GIS Cut Line= 3
      1607617.91      6811200.49      1608631.99      6812261.77
      1609265.01      6813003.76
#Sta/Elev= 30
  3520.5 1801.07  3629.7 1798.56  3773.5  1792.3  3890.6 1790.34  3933.9 1790.28
  3997.7 1786.94  4047.1 1786.25  4068.5 1790.21  4089.5 1791.87  4485.5 1791.64
  4733.4  1789.8  4902.9 1790.99  4938.4 1788.16  4973.6 1788.77  4986.9 1781.66
  5001.6 1780.39  5003.1 1779.89  5017.6 1780.39  5037.1 1790.01  5051.3 1791.16
  5229.2 1789.38  5292.9 1784.57  5321.4 1783.98  5374.1 1786.58  5396.6 1786.11
    5406 1785.89  5427.9    1790  5448.8  1791.9  5561.9 1795.89  5963.7 1797.83
#Mann= 7 ,-1 , 0
  3520.5     .05       0  3773.5     .12       0  3890.6     .05       0
  5001.6    .035       0  5017.6     .05       0  5374.1     .12       0
  5396.6     .05       0
Bank Sta=5001.6,5017.6
XS Rating Curve= 0 ,0
Exp/Cntr=0.3,0.1

Type RM Length L Ch R = 1 ,51397   ,580,580,580
BEGIN DESCRIPTION:
Lytle Creek 52085.131
END DESCRIPTION:
XS GIS Cut Line= 4
      1607058.67      6812453.32      1607904.32      6812837.79
      1608143.83      6812940.44      1609091.22      6812913.24
#Sta/Elev= 30
  4073.2 1790.49  4579.9 1790.37    4626 1786.87  4723.8 1782.86  4752.3 1783.25
  4775.4 1785.56  4890.7 1787.38  4965.4 1786.24  4980.9 1782.05  4999.8 1780.85
  5017.3 1781.67  5024.6 1785.46  5035.4 1786.51  5093.4 1787.71    5604 1787.65
    5634 1787.33  5642.1 1780.46  5643.6 1779.96  5658.1 1780.46  5664.1  1786.9
  5675.8 1786.99  5704.1  1786.9  5744.1 1780.41  5754.1 1780.25  5774.9 1784.93
  5794.1 1786.92  5824.1 1785.96  5869.8 1789.01  6044.2 1795.01  6210.5 1796.68
#Mann= 5 ,-1 , 0
  4073.2     .05       0  5642.1     .05       0  5658.1     .05       0
  5675.8     .12       0  5774.9     .05       0
Bank Sta=5642.1,5658.1
XS Rating Curve= 0 ,0
Exp/Cntr=0.3,0.1

Type RM Length L Ch R = 1 ,50817   ,422,422,422
BEGIN DESCRIPTION:
Lytle Creek 51500.99
END DESCRIPTION:
XS GIS Cut Line= 3
      1606769.64      6812838.68      1607677.77      6813314.43
      1609389.49      6813901.21
#Sta/Elev= 30
  3974.8 1789.81  4453.8 1789.83  4652.3 1785.87  4816.2 1785.85  4861.4 1784.03
  4940.4 1786.02  4969.2 1784.45  4998.5  1775.9  5010.2 1775.16  5011.7 1774.66
  5026.2 1775.16  5039.4 1781.55  5056.2 1786.11  5134.5 1786.74  5207.3 1785.31
  5229.6 1782.93  5243.9  1778.8  5261.2 1779.55  5269.9 1781.61  5314.2 1782.86
  5483.4  1785.3  5546.1 1787.43  5927.3 1787.64  6064.8 1791.08  6140.3 1796.23
  6159.9 1795.16  6191.6 1795.87    6380 1801.94  6656.2 1807.07  6809.5 1807.79
#Mann= 5 ,-1 , 0
  3974.8     .05       0  4969.2     .12       0  5010.2     .07       0
  5026.2     .12       0  5261.2     .05       0
Bank Sta=5010.2,5026.2
XS Rating Curve= 0 ,0
Exp/Cntr=0.3,0.1

Type RM Length L Ch R = 1 ,50395   ,659,659,659
BEGIN DESCRIPTION:
Lytle Creek 50902.465
END DESCRIPTION:
XS GIS Cut Line= 3
      1606925.66      6813047.83      1607513.26       6813686.2
      1608435.94      6814527.23
#Sta/Elev= 30
    4147 1789.61  4373.2 1788.76  4578.5 1783.56    4642 1783.41  4649.4 1782.76
  4790.6 1783.19  4818.9 1782.35  4826.3 1780.57  4833.1 1781.19  4838.6 1777.94
  4840.1 1777.44  4855.9 1777.94  4861.5 1779.17  4875.6 1780.08  4896.6 1780.14
    4904 1781.29  4918.2 1781.47  4965.5 1779.08  4989.1 1778.88  5095.2 1783.28
  5130.3 1782.03  5165.8 1782.01  5215.4 1782.75  5250.6 1784.39  5335.7 1785.09
  5696.5 1783.61  5767.5 1784.18  5965.4  1794.2  6128.3 1799.55  6263.1 1801.51
#Mann= 3 ,-1 , 0
    4147     .05       0  4838.6     .05       0  4855.9     .05       0
Bank Sta=4838.6,4855.9
XS Rating Curve= 0 ,0
Exp/Cntr=0.3,0.1

Type RM Length L Ch R = 1 ,49736   ,437,437,437
BEGIN DESCRIPTION:
Lytle Creek 50408.91
END DESCRIPTION:
XS GIS Cut Line= 3
      1606643.27      6813785.65      1607153.65      6814066.88
      1607875.81      6814569.52
#Sta/Elev= 30
  4442.2 1787.71  4497.2 1789.48  4578.6 1790.29  4665.7 1788.79  4718.2 1789.05
  4806.8 1784.82    4856 1780.97  4866.4 1778.12  4872.1 1777.73  4909.9 1779.15
  4969.4 1779.71  4975.3 1776.02    4981 1776.05    4995 1769.95  4996.5 1769.45
  5012.3 1769.95  5018.8 1770.61  5022.8 1774.12  5028.8 1774.12  5034.2 1778.57
    5049 1780.28  5069.9 1781.53  5138.9 1782.24  5564.8 1782.28  5594.5 1782.82
  5623.6 1785.07    5687 1787.47  5794.3  1787.8  5809.1 1787.02  5904.8 1789.67
#Mann= 4 ,-1 , 0
  4442.2     .05       0    4995    .035       0  5012.3     .05       0
  5138.9     .05       0
Bank Sta=4995,5012.3
XS Rating Curve= 0 ,0
Exp/Cntr=0.3,0.1

Type RM Length L Ch R = 1 ,49299   ,478,478,478
BEGIN DESCRIPTION:
Lytle Creek 49971.07
END DESCRIPTION:
XS GIS Cut Line= 3
      1606643.23      6814167.57      1606959.21      6814438.41
      1607358.49      6814785.61
#Sta/Elev= 30
  4557.6 1783.94  4644.2 1782.95  4672.7 1783.56  4750.6 1781.78    4800 1781.74
  4828.6 1780.69  4857.1 1778.37  4885.6 1778.02  4906.5 1775.11  4914.2 1775.45
  4920.7 1777.59  4937.3  1777.8  4963.6 1777.49  4969.6  1775.8  4973.8  1775.8
  4977.8 1773.31    4990 1772.63  4991.5 1772.13  5007.3 1772.63  5020.5 1773.65
  5027.2 1775.04  5034.5 1777.81  5106.5 1779.81  5168.6 1781.03  5254.1 1780.74
  5346.2  1778.2  5352.8 1778.44  5381.3 1784.17  5459.2 1789.83  5502.9  1790.8
#Mann= 5 ,-1 , 0
  4557.6     .05       0  4937.3     .12       0    4990     .07       0
  5007.3     .12       0  5106.5     .05       0
Bank Sta=4990,5007.3
XS Rating Curve= 0 ,0
Exp/Cntr=0.3,0.1

Type RM Length L Ch R = 1 ,48821   ,432,432,432
BEGIN DESCRIPTION:
Lytle Creek 49573.62
END DESCRIPTION:
XS GIS Cut Line= 3
      1606513.22      6814197.15      1606499.24      6814512.75
      1607014.77      6815379.39
#Sta/Elev= 30
  4327.4 1783.22  4428.4 1783.41  4538.5 1781.39  4835.1 1780.25  4899.3 1778.94
  4973.4 1776.18  4994.8 1771.82  5016.2 1774.22    5022 1773.17  5023.1 1770.83
  5024.6 1770.33  5040.4 1770.83    5045 1773.09  5068.3 1774.06  5080.4 1775.67
  5090.2 1775.02    5096 1771.79  5103.2 1771.54  5111.6 1772.06  5117.4 1775.32
    5133 1774.57  5184.7  1777.2  5219.6 1773.48  5228.5 1773.71  5234.3 1774.55
  5255.7  1780.9  5271.3 1783.11    5431 1793.16  5526.5 1795.79  5651.7 1797.15
#Mann= 3 ,-1 , 0
  4327.4     .05       0  5023.1     .05       0  5040.4     .05       0
Bank Sta=5023.1,5040.4
XS Rating Curve= 0 ,0
Exp/Cntr=0.3,0.1

Type RM Length L Ch R = 1 ,48389   ,377,377,377
BEGIN DESCRIPTION:
Lytle Creek 49035.02
END DESCRIPTION:
XS GIS Cut Line= 3
      1606542.45      6813939.37      1606362.38      6814924.01
       1606466.1       6815653.3
#Sta/Elev= 30
    3797 1785.46  3876.9 1783.21  4009.1 1783.14  4033.7 1781.85  4086.9 1782.24
    4092 1781.22  4161.6 1781.29  4192.1 1782.54  4203.5 1781.08  4242.9 1781.79
  4862.6 1777.98    4903 1778.66  4913.1 1778.08  4933.3 1774.96  4953.5 1774.15
  4963.6 1771.71  4983.8 1769.43    5004 1769.33  5014.1 1768.25  5015.6 1766.87
  5017.1 1766.37  5032.9 1766.87  5062.4 1773.38  5074.7 1772.94    5105  1775.1
  5145.4 1780.02  5236.3 1784.08  5357.5 1787.37  5416.7 1786.53  5534.6 1786.62
#Mann= 3 ,-1 , 0
    3797     .05       0  5015.6     .05       0  5032.9     .05       0
Bank Sta=5015.6,5032.9
XS Rating Curve= 0 ,0
Exp/Cntr=0.3,0.1

Type RM Length L Ch R = 1 ,48012   ,507,507,507
BEGIN DESCRIPTION:
Lytle Creek 48676.464
END DESCRIPTION:
XS GIS Cut Line= 3
      1606569.59      6813740.04       1606021.8      6815023.04
      1606045.15      6815797.54
#Sta/Elev= 30
  3440.2 1785.28  3564.8 1785.09  3717.3 1782.19  4362.2 1780.76  4432.6 1779.93
  4456.2 1778.63  4503.4 1778.28  4547.1 1778.15  4608.7 1779.13  4775.4 1777.99
  4840.2 1778.32  4870.2 1777.74  4914.8    1775  4960.3 1772.52  4980.3 1768.66
  4990.3 1767.55  4991.6 1766.44  4993.1 1765.94  5008.9 1766.44  5010.3 1767.31
  5022.9 1770.34  5030.3 1771.61  5070.3  1772.3  5140.3 1778.44  5170.4 1780.33
  5210.4 1782.32  5230.4 1782.43  5270.4 1784.02  5350.4 1785.83  5610.1  1785.4
#Mann= 5 ,-1 , 0
  3440.2     .05       0  4914.8     .12       0  4991.6     .07       0
  5008.9     .12       0  5022.9     .05       0
Bank Sta=4991.6,5008.9
XS Rating Curve= 0 ,0
Exp/Cntr=0.3,0.1

Type RM Length L Ch R = 1 ,47505   ,807,807,807
BEGIN DESCRIPTION:
Mapping XS 1c9a4dce
END DESCRIPTION:
XS GIS Cut Line= 4
      1604820.01      6814331.81      1605255.39      6814628.19
      1605738.43      6815768.98      1605998.33      6815969.02
#Sta/Elev= 30
  3721.3 1785.86  3751.5  1784.4    3887 1780.69  4009.7 1778.69  4414.9 1777.46
  4515.1 1776.25  4627.9 1775.87  4703.9 1776.64  4714.7 1776.14  4879.2 1776.45
  4902.9 1775.71  4921.1 1773.83  4926.6  1772.9    4932 1770.93  4964.5 1767.94
  4973.9 1767.92  4988.3 1765.83  4989.8 1765.33  5005.9 1765.83  5073.1 1769.48
  5103.2    1773  5149.1 1775.95  5232.5  1779.5  5332.6 1779.84  5420.6 1782.43
  5497.4 1782.19  5561.8 1784.05  5690.4  1784.2  5783.8 1785.99  5814.8 1785.97
#Mann= 3 ,-1 , 0
  3721.3     .05       0  4988.3     .05       0  5005.9     .05       0
Bank Sta=4988.3,5005.9
XS Rating Curve= 0 ,0
Exp/Cntr=0.3,0.1

Type RM Length L Ch R = 1 ,46698   ,475,475,475
BEGIN DESCRIPTION:
Lytle Creek 47289.81
END DESCRIPTION:
XS GIS Cut Line= 3
      1604504.39      6814757.78      1604876.98        6815744.
      1605729.62      6816032.26
#Sta/Elev= 30
  4158.4 1783.94  4174.5 1784.25  4190.7 1782.05  4204.7 1782.31  4212.1 1783.98
  4314.7 1777.59  4468.6 1774.05  4545.5 1774.49  4554.2 1776.25  4570.3 1773.44
  4630.7 1773.87  4735.4 1771.37  4801.1 1774.55  4898.3 1774.72  4941.3 1774.09
  4960.4 1772.06  4982.2 1761.77  4983.7 1761.27  4999.8 1761.77  5013.8 1762.26
  5035.2 1768.88  5064.2 1771.31  5206.2 1774.09  5369.9 1772.27  5421.7 1773.66
  5453.4 1776.84    5459 1775.14  5495.7 1774.96  5780.6 1780.37  6112.7 1783.42
#Mann= 5 ,-1 , 0
  4158.4     .05       0  4898.3     .12       0  4982.2     .07       0
  4999.8     .12       0  5064.2     .05       0
Bank Sta=4982.2,4999.8
XS Rating Curve= 0 ,0
Exp/Cntr=0.3,0.1

Type RM Length L Ch R = 1 ,46223   ,425,425,425
BEGIN DESCRIPTION:
Lytle Creek 46784.46
END DESCRIPTION:
XS GIS Cut Line= 4
      1603874.69      6815088.92      1604305.57      6815723.05
      1604401.95      6815758.99      1605901.02      6816138.96
#Sta/Elev= 30
  4128.3 1777.31  4163.5  1775.8  4192.4  1776.5    4502 1773.63  4951.9 1773.12
  4958.4  1772.7  4969.1 1769.34  4977.5 1764.68  4982.9 1763.63  4987.9  1760.3
  4989.4  1759.8  5005.7  1760.3  5021.6 1763.85  5031.9 1768.04  5042.2 1769.44
  5097.3 1769.74  5142.3 1773.05  5289.8 1774.59    5379 1774.33  5460.9 1771.95
  5630.3 1771.83  5754.1 1773.75  5783.7  1775.7  5788.8 1774.92  5795.3 1776.24
  5829.8  1775.1  5888.2 1777.56  6022.3 1780.31  6434.2 1783.85  6544.3 1783.57
#Mann= 5 ,-1 , 0
  4128.3     .05       0  4951.9     .12       0  4987.9     .07       0
  5005.7     .12       0  5142.3     .05       0
Bank Sta=4987.9,5005.7
XS Rating Curve= 0 ,0
Exp/Cntr=0.3,0.1

Type RM Length L Ch R = 1 ,45798   ,480,480,480
BEGIN DESCRIPTION:
Lytle Creek 46259.37
END DESCRIPTION:
XS GIS Cut Line= 3
      1603650.13      6816087.52      1604514.03      6816197.52
      1605770.83      6816154.85
#Sta/Elev= 30
  4272.3 1785.25  4297.4 1785.44  4314.1 1782.63  4473.9 1774.85    4751 1767.89
  4788.5 1770.54  4831.6 1769.65  4882.1 1763.53  4902.2  1764.1  4922.4 1768.74
  4953.4 1771.11  4972.8 1763.06  4991.6 1761.94  4994.1 1761.78  4995.6 1761.28
  5011.9 1761.78  5033.3 1763.15  5063.5 1773.27  5134.1 1772.17  5244.2 1772.56
  5344.3 1768.75  5424.3  1772.7  5594.4 1770.45  5804.5 1772.51  5854.6 1774.44
  5867.7 1776.77  5874.6 1775.18  5904.6 1775.48  6184.7  1782.1  6400.7 1782.88
#Mann= 5 ,-1 , 0
  4272.3     .05       0  4991.6     .12       0  4994.1     .07       0
  5011.9     .12       0  5134.1     .05       0
Bank Sta=4994.1,5011.9
XS Rating Curve= 0 ,0
Exp/Cntr=0.3,0.1

Type RM Length L Ch R = 1 ,45318   ,356,356,356
BEGIN DESCRIPTION:
Lytle Creek 45801.99
END DESCRIPTION:
XS GIS Cut Line= 3
      1603894.01      6816807.53      1604623.89      6816591.54
      1605607.03       6816228.2
#Sta/Elev= 30
  4367.1 1777.71  4639.3 1773.15  4770.2 1772.63  4808.7 1773.56  4875.2 1772.62
  4880.4 1771.05  4908.4 1771.01  4920.8 1769.57  4962.6  1768.4    4973 1763.05
  4980.2 1760.93  4995.4 1759.26  4996.9 1758.76  5013.2 1759.26  5036.7 1761.69
    5046 1762.66  5051.9 1766.06  5066.9 1771.51  5077.3 1772.68  5188.8 1771.46
  5246.7 1770.13  5387.2 1770.69  5442.7 1769.43  5598.5 1771.15  5755.9 1771.33
  5816.7 1773.19  5847.2 1776.31  5877.6 1775.45  5982.3 1780.21  6176.4 1782.07
#Mann= 5 ,-1 , 0
  4367.1     .05       0  4995.4     .05       0  5013.2     .05       0
  5036.7     .12       0  5188.8     .05       0
Bank Sta=4995.4,5013.2
XS Rating Curve= 0 ,0
Exp/Cntr=0.3,0.1

Type RM Length L Ch R = 1 ,44962   ,566,566,566
BEGIN DESCRIPTION:
Mapping XS 67b3d247
END DESCRIPTION:
XS GIS Cut Line= 5
      1603680.72      6817099.03       1604573.8      6817082.22
      1604756.84      6816822.69      1605408.05      6816562.77
      1605637.23       6816444.7
#Sta/Elev= 30
  3923.1 1780.19  4017.4 1777.47    4243 1773.35  4357.5 1773.55  4427.5 1772.16
  4597.5 1772.08  4827.4 1769.89  4892.7 1771.19  4943.2 1769.65  4956.1 1767.93
  4970.2 1763.56  4990.9 1760.36  4992.4 1759.86  5008.7 1760.36  5041.8 1762.02
  5050.3 1763.56  5056.4  1766.2  5065.1 1768.19  5084.8 1769.95  5115.2 1771.14
  5172.2 1770.05  5196.5  1769.1  5698.4 1769.83    5821 1774.23  5834.8 1777.29
  5865.4 1775.07  5874.6 1775.21  5896.8 1778.02  5946.8 1779.46  6092.9 1780.52
#Mann= 5 ,-1 , 0
  3923.1     .05       0  4990.9     .05       0  5008.7     .05       0
  5084.8     .12       0  5172.2     .05       0
Bank Sta=4990.9,5008.7
XS Rating Curve= 0 ,0
Exp/Cntr=0.3,0.1

Type RM Length L Ch R = 1 ,44396   ,231,231,231
BEGIN DESCRIPTION:
Mapping XS 19fa8d52
END DESCRIPTION:
XS GIS Cut Line= 4
        1603814.      6817190.13      1604466.58      6817264.11
      1605810.83      6817038.46      1605998.36      6817017.63
#Sta/Elev= 30
  3654.3 1775.37  3786.1 1773.29  3896.8 1773.56  4088.1 1770.57  4390.6 1770.14
  4461.6 1768.18  4512.3 1769.88  4542.7 1768.65  4664.3 1769.69  4856.7 1766.21
  4897.6 1764.25  4917.3 1761.96  4922.4 1763.35  4938.1 1760.48  4974.1 1758.64
  4975.6 1758.14  4991.9 1758.64  5029.4 1759.79  5038.5 1762.39  5043.6 1761.44
  5049.7 1764.41  5059.8 1766.91  5080.1 1769.97  5104.2    1770  5225.5    1775
  5252.5 1778.54  5445.1 1782.88  5658.1 1781.96  5839.3 1784.81  5862.8 1784.26
#Mann= 3 ,-1 , 0
  3654.3     .05       0  4974.1     .05       0  4991.9     .05       0
Bank Sta=4974.1,4991.9
XS Rating Curve= 0 ,0
Exp/Cntr=0.3,0.1

Type RM Length L Ch R = 1 ,44165   ,288,288,288
BEGIN DESCRIPTION:
Lytle Creek 44695.53
END DESCRIPTION:
XS GIS Cut Line= 3
      1603652.26      6817201.89       1605050.6      6817358.02
      1605870.47      6817462.24
#Sta/Elev= 30
    3591 1778.91  3714.5 1775.48  3865.4 1773.27  3986.2 1773.51  4056.6 1771.48
  4096.9 1771.88  4167.3  1770.5  4308.2 1770.92  4459.1 1769.73  4559.7 1767.66
  4678.9 1769.17    4932 1768.89    4955 1766.46  4962.2 1762.62  4982.3 1758.08
  5003.6  1756.6  5005.1  1756.1  5021.4  1756.6  5022.6 1758.34  5037.7 1759.75
    5063 1767.29  5083.1 1772.26  5112.6 1775.25  5117.6 1774.81  5133.5 1775.98
  5197.6 1776.95  5244.4 1779.43    5315 1781.68  5357.5 1780.66  5824.5  1783.5
#Mann= 3 ,-1 , 0
    3591     .05       0  5003.6     .05       0  5021.4     .05       0
Bank Sta=5003.6,5021.4
XS Rating Curve= 0 ,0
Exp/Cntr=0.3,0.1

Type RM Length L Ch R = 1 ,43877   ,385,385,385
BEGIN DESCRIPTION:
Lytle Creek 44398.8
END DESCRIPTION:
XS GIS Cut Line= 4
      1603842.25        6817315.      1604282.96      6817556.21
      1605003.73      6817639.27      1605426.59      6817722.97
#Sta/Elev= 30
  3782.6 1773.21  3822.9 1773.32  3882.6  1772.1  3964.2 1772.28  4073.2  1769.4
  4176.6  1768.2  4432.3 1767.89  4538.7 1766.32  4610.3 1767.28  4689.2 1767.12
    4740 1768.01  4911.2 1767.31  4951.1 1768.46  4961.5 1766.24  4971.6 1760.09
  4981.6 1755.79  4982.8 1754.46  4984.3 1753.96  4999.1 1753.96  5000.6 1754.46
  5013.7 1754.82  5028.4 1761.16  5042.4 1762.13  5062.8 1769.08    5073 1771.64
  5093.4 1773.72  5225.9 1774.42  5387.1 1778.57  5409.4 1778.06  5441.6  1778.5
#Mann= 3 ,-1 , 0
  3782.6     .05       0  4982.8     .05       0  5000.6     .05       0
Bank Sta=4982.8,5000.6
XS Rating Curve= 0 ,0
Exp/Cntr=0.3,0.1

Type RM Length L Ch R = 1 ,43492   ,381,381,381
BEGIN DESCRIPTION:
Lytle Creek 44192.169
END DESCRIPTION:
XS GIS Cut Line= 3
      1604052.97      6817641.21      1604959.74      6818022.54
      1605369.84      6817901.08
#Sta/Elev= 30
  4023.6 1768.74  4123.4 1767.34  4212.2 1767.94    4236 1766.54  4242.8 1767.28
  4336.4 1767.28  4341.8 1766.54  4427.2 1765.81  4624.7    1765  4772.6 1767.39
  4861.1 1766.45  4902.2 1767.35  4937.1  1762.8  4955.1 1756.57  4984.3 1757.54
  4993.1  1756.3  4994.6  1755.8  5010.9  1756.3  5033.6 1756.94  5039.9 1760.56
  5045.1 1759.15  5064.9 1768.97  5183.3 1770.24  5283.1 1772.99  5294.4 1774.47
  5346.5  1774.5  5367.4 1776.21  5409.1 1776.69  5426.5 1774.68    5435 1775.07
#Mann= 3 ,-1 , 0
  4023.6     .05       0  4993.1     .05       0  5010.9     .05       0
Bank Sta=4993.1,5010.9
XS Rating Curve= 0 ,0
Exp/Cntr=0.3,0.1

Type RM Length L Ch R = 1 ,43111   ,505,505,505
BEGIN DESCRIPTION:
Lytle Creek 43609.297
END DESCRIPTION:
XS GIS Cut Line= 3
      1603804.11       6817832.1      1604790.35      6818351.95
      1605720.51      6818758.28
#Sta/Elev= 30
  3863.7 1775.12    3912 1775.44    4023 1773.51  4060.6  1774.1    4077 1772.01
  4187.1 1763.93  4305.6 1762.44  4357.7 1762.47  4429.9 1764.36  4594.3 1764.08
  4764.9 1766.62  4808.9 1768.85  4814.6 1767.23  4847.3 1763.26    4897 1764.42
  4913.4 1758.18  4919.1 1757.46  4941.1 1761.16  4978.4  1759.2  4994.5 1753.64
  4999.6 1753.64  5001.1 1753.14  5017.5 1753.64  5031.9 1753.81  5049.1 1756.69
  5060.8 1764.33  5070.9 1767.21  5206.7 1766.22  5485.9 1767.05  5993.6 1779.32
#Mann= 3 ,-1 , 0
  3863.7     .05       0  4999.6     .05       0  5017.5     .05       0
Bank Sta=4999.6,5017.5
XS Rating Curve= 0 ,0
Exp/Cntr=0.3,0.1

Type RM Length L Ch R = 1 ,42606   ,403,403,403
BEGIN DESCRIPTION:
Lytle Creek 43080.136
END DESCRIPTION:
XS GIS Cut Line= 3
      1603756.59      6817854.29      1604389.76      6818626.28
      1605635.22      6819373.59
#Sta/Elev= 30
  3994.8 1776.23    4110 1776.84  4245.3 1774.33    4273 1771.94  4295.2 1771.75
  4336.8 1766.58  4400.7  1762.7  4465.2 1760.99  4550.7 1761.53  4614.5 1763.26
  4727.9 1762.92  4898.7 1764.26  4962.6 1766.55  4969.6  1765.6    4977 1760.96
  4990.4 1750.01  4991.9 1749.51  5008.3 1750.01  5011.6 1753.95  5034.3 1754.73
  5079.6 1761.59  5085.4 1764.15    5101 1765.13  5159.3 1764.29  5186.5 1765.49
  5668.5 1763.91  5827.9 1764.56  6171.9 1767.97  6214.7 1769.89  6445.7 1775.14
#Mann= 3 ,-1 , 0
  3994.8     .05       0  4990.4     .05       0  5008.3     .05       0
Bank Sta=4990.4,5008.3
XS Rating Curve= 0 ,0
Exp/Cntr=0.3,0.1

Type RM Length L Ch R = 1 ,42203   ,1287,1287,1287
BEGIN DESCRIPTION:
Lytle Creek 42668.9
END DESCRIPTION:
XS GIS Cut Line= 5
      1603626.54      6818050.53      1604184.22      6818932.76
      1604303.93      6819021.54      1604480.59      6819130.83
      1605399.85      6819268.56
#Sta/Elev= 30
  3819.7 1777.05  4018.5 1774.16  4146.9 1767.54  4185.6 1765.94  4194.9 1762.37
  4200.8 1762.28  4216.1 1753.44  4240.9 1751.17  4273.8 1751.11  4301.7 1761.54
  4346.7  1767.8  4352.6 1767.86  4367.9 1762.46  4396.4 1761.81    4796 1763.56
  4902.7 1765.92  4939.1 1764.66  4967.4 1757.13  4975.8 1751.87  4988.9  1748.4
  5001.1 1747.58  5002.6 1747.08    5019 1747.58  5025.5 1748.53  5032.8 1754.67
  5038.7 1753.62  5048.2 1761.19  5060.7 1764.44  5699.9 1763.06  6149.7 1769.45
#Mann= 5 ,-1 , 0
  3819.7     .05       0  4146.9     .12       0  4240.9     .05       0
  5001.1     .05       0    5019     .05       0
#XS Ineff= 2 , 0
       0    4354 1772.09               0
Permanent Ineff=
       F       F
Bank Sta=5001.1,5019
XS Rating Curve= 0 ,0
Exp/Cntr=0.3,0.1

Type RM Length L Ch R = 1 ,40916   ,867,867,867
BEGIN DESCRIPTION:
Lytle Creek 40789.027
END DESCRIPTION:
XS GIS Cut Line= 4
       1603546.7      6817961.58      1603778.14      6818679.26
      1604072.72      6819508.53      1605129.21       6820029.1
#Sta/Elev= 30
    2485 1776.01  2701.9 1776.06  2901.5 1769.75  2943.6 1765.49  2975.1 1753.85
  3002.2 1753.83  3078.6 1753.76  3115.9 1766.85  3122.2 1767.06  3132.7 1761.85
    3164 1760.84  3906.7 1763.25  4605.5 1762.31  4679.1 1765.45  4723.7 1756.11
  4745.9 1754.99  4768.3 1754.82  4830.1 1760.38  4925.5 1758.88  4980.1 1753.19
  4987.3  1751.4    4990 1746.26    4992 1745.76    5010 1746.26  5015.3 1751.41
  5032.2 1757.35  5060.3 1759.61  5077.1 1766.21  5091.5 1768.61  5296.9 1775.69
#Mann= 5 ,-1 , 0
    2485     .05       0  3002.2     .12       0    3164     .05       0
    4990     .05       0    5010     .05       0
#XS Ineff= 2 , 0
       0  3115.3 1771.78               0
Permanent Ineff=
       F       F
Bank Sta=4990,5010
XS Rating Curve= 0 ,0
Exp/Cntr=0.3,0.1

Type RM Length L Ch R = 1 ,40049   ,808,808,808
BEGIN DESCRIPTION:
Lytle Creek 40238.718
END DESCRIPTION:
XS GIS Cut Line= 4
      1603472.83      6818104.19      1603547.41      6818993.46
      1604007.72      6819608.81      1604496.13       6820697.4
#Sta/Elev= 30
  2824.1 1775.59  3018.6 1773.28    3129 1769.39  3209.3 1763.48  3249.4 1750.47
  3270.5 1749.25  3339.7 1752.08  3359.8 1760.73  3401.6 1763.83    3430 1764.65
  3460.1 1759.22  4118.5 1762.29  4418.6 1761.36  4460.3 1763.08  4761.4 1760.02
  4901.8 1761.65  4944.4 1760.65  4952.3 1753.54  4966.3 1750.94  4966.5 1748.36
    4968 1747.86  4984.5 1748.36  5010.2 1751.42  5028.1  1750.8  5102.3 1753.52
  5200.5 1750.79  5218.2 1757.81  5246.8 1762.85    5345 1772.53  5678.1 1777.98
#Mann= 7 ,-1 , 0
  2824.1     .05       0  3270.5     .12       0  3401.6     .05       0
  4901.8     .12       0  4966.5     .07       0  4984.5     .12       0
  5028.1     .05       0
#XS Ineff= 2 , 0
       0  3424.4 1768.73  6575.6       0 1768.73
Permanent Ineff=
       F       F
Bank Sta=4966.5,4984.5
XS Rating Curve= 0 ,0
Exp/Cntr=0.3,0.1

Type RM Length L Ch R = 1 ,39241   ,597,597,597
BEGIN DESCRIPTION:
Lytle Creek 39640.856
END DESCRIPTION:
XS GIS Cut Line= 3
      1602408.27      6818826.06      1603733.34       6820036.1
      1604269.62      6820631.84
#Sta/Elev= 30
  3329.8 1769.31  3420.6 1765.84  3845.5 1759.89  4093.5 1753.42  4114.4 1754.55
    4157  1752.5  4178.5 1754.64  4206.3 1753.54  4291.4  1757.2  4539.3 1759.41
  4638.6 1758.15  4893.4 1760.85  4928.5 1758.61  4950.1 1752.32  4971.1 1749.79
    4983  1743.7  4984.5  1743.2    5001  1743.7  5020.4 1749.28  5070.4 1757.33
  5105.5 1759.02  5275.1 1762.49  5353.6 1759.42  5402.9 1759.29  5544.2 1765.24
  5608.5 1769.92  5643.6 1769.44  5657.8 1770.27    5672 1773.22  5925.8 1777.45
#Mann= 3 ,-1 , 0
  3329.8     .05       0    4983     .05       0    5001     .05       0
Bank Sta=4983,5001
XS Rating Curve= 0 ,0
Exp/Cntr=0.3,0.1

Type RM Length L Ch R = 1 ,38644   ,961,961,961
BEGIN DESCRIPTION:
Lytle Creek 39054.887
END DESCRIPTION:
XS GIS Cut Line= 3
      1601558.89      6820051.98      1603813.71      6820547.04
      1604131.36      6820607.03
#Sta/Elev= 30
  2807.2  1789.1  2936.3 1786.43  3044.5 1770.06  3120.6 1764.43  3322.6 1759.36
  3698.5 1754.55  3796.3 1749.77  4210.9 1756.19  4420.9 1757.45  4440.1 1757.79
  4445.3 1759.15  4922.5 1759.46    4943 1755.21  4957.7 1754.34  4973.7 1749.86
    4984 1744.51  4991.7 1743.17  5005.7 1741.73  5007.2 1741.23  5023.7 1741.73
  5035.1 1747.67  5045.3 1759.04  5106.8 1757.63  5160.1 1759.64  5202.6 1760.03
    5255 1763.78  5260.1 1762.72    5290 1766.51  5330.8 1765.63    5439 1773.25
#Mann= 5 ,-1 , 0
  2807.2     .05       0  4991.7     .12       0  5005.7     .07       0
  5023.7     .12       0  5160.1     .05       0
Bank Sta=5005.7,5023.7
XS Rating Curve= 0 ,0
Exp/Cntr=0.3,0.1

Type RM Length L Ch R = 1 ,37683   ,644,644,644
BEGIN DESCRIPTION:
Lytle Creek 38501.12
END DESCRIPTION:
XS GIS Cut Line= 3
      1601730.45      6820565.33      1603565.73      6821530.52
      1604784.68      6821084.78
#Sta/Elev= 30
  2572.1 1773.47  2828.2 1770.85  2894.3 1767.42  3015.2 1756.19  3163.9 1752.19
  3243.9 1755.31  3279.7 1752.31  3435.9 1751.44  3466.8 1756.93  3488.8 1752.12
  3516.5 1751.66  4586.3 1755.39  4830.3 1756.37  4858.3 1756.52  4921.8 1757.01
  4958.9 1753.28  4964.4 1749.11    4975 1744.94  4987.3 1742.28  4988.8 1741.78
  5005.3 1742.28  5028.2 1744.18  5038.9  1748.4  5045.2 1753.47  5071.3 1755.28
  5113.4 1757.24  5309.3 1757.31  5613.9 1771.97  5784.2  1776.8  5943.6 1777.61
#Mann= 7 ,-1 , 0
  2572.1     .05       0  4586.3     .12       0  4830.3     .05       0
  4858.3     .12       0  4987.3     .07       0  5005.3     .12       0
  5071.3     .05       0
Bank Sta=4987.3,5005.3
XS Rating Curve= 0 ,0
Exp/Cntr=0.3,0.1

Type RM Length L Ch R = 1 ,37039   ,730,730,730
BEGIN DESCRIPTION:
Lytle Creek 37390.876
END DESCRIPTION:
XS GIS Cut Line= 4
      1601666.63      6820635.33      1603591.54      6821990.04
      1604013.02      6822041.39      1604701.25      6822163.51
#Sta/Elev= 30
  2228.5 1773.17  2487.2 1769.41  2567.4 1770.23  2680.6 1758.42  2975.1 1751.03
  3155.9  1750.6  3191.9 1756.41  3227.7 1758.02  3263.4 1751.27  3391.4 1750.48
  4298.2 1754.47  4535.6    1754  4858.9 1755.25  4908.2 1751.77  4935.5  1751.8
  4940.5 1749.79  4948.5 1752.29  4958.5  1751.8  4968.6 1746.23  4979.8 1745.81
  4981.3 1745.31  4997.8 1745.81  5039.4 1746.94  5049.6 1748.15  5069.1 1755.19
  5074.2 1754.16  5100.3 1757.59  5151.1 1753.45    5273 1762.88  5705.9 1771.22
#Mann= 5 ,-1 , 0
  2228.5     .05       0  4298.2     .12       0  4535.6     .05       0
  4979.8     .05       0  4997.8     .05       0
Bank Sta=4979.8,4997.8
XS Rating Curve= 0 ,0
Exp/Cntr=0.3,0.1

Type RM Length L Ch R = 1 ,36309   ,1306,1306,1306
BEGIN DESCRIPTION:
Lytle Creek 36844.86
END DESCRIPTION:
XS GIS Cut Line= 3
      1601707.74       6821526.3      1603091.84      6822112.36
      1603983.04      6823023.65
#Sta/Elev= 30
  2865.1 1760.82  3068.5 1754.79  3603.2 1748.83  3650.6 1746.47  3741.7 1748.64
  4402.7 1751.64  4473.5  1748.3  4494.6 1751.13    4537 1753.03  4579.5 1751.39
  4671.3 1753.57  4738.3 1751.25  4839.3 1752.45  4883.5 1751.83  4918.9 1749.56
  4925.9  1747.5  4933.1 1748.84  4940.1 1744.51  4954.2 1745.34  4966.5 1744.18
    4968 1743.68  4984.5 1744.18  5039.1 1745.41  5060.4 1755.13  5074.5 1759.49
  5131.1 1763.37  5152.3 1762.51  5180.5 1764.56  5392.7 1764.29  5642.8 1766.88
#Mann= 5 ,-1 , 0
  2865.1     .05       0  4738.3     .12       0  4839.3     .05       0
  4966.5     .05       0  4984.5     .05       0
Bank Sta=4966.5,4984.5
XS Rating Curve= 0 ,0
Exp/Cntr=0.3,0.1

Type RM Length L Ch R = 1 ,35003   ,884,884,884
BEGIN DESCRIPTION:
Lytle Creek 35725.689
END DESCRIPTION:
XS GIS Cut Line= 4
      1601443.58      6822204.53      1602476.76      6822941.71
      1602982.34      6823477.08      1603657.43      6823092.95
#Sta/Elev= 30
  3276.9 1772.77  3552.4 1768.51  3632.3 1764.34  3795.8 1749.46  3982.6 1744.61
  4026.8 1747.81  4133.8 1749.45  4744.9 1749.36  4959.6 1748.24  4966.9 1747.53
  4973.7 1744.05    4981 1736.61  4985.9 1735.29  4987.4 1734.79  5003.9 1735.29
  5023.1 1738.94  5030.4 1744.09  5051.4  1746.9  5093.9 1746.08  5123.3 1739.55
  5136.4 1740.38  5143.7 1743.57  5150.5 1742.68  5164.7 1747.68  5242.5 1751.08
  5456.2 1749.27    5647 1748.96  5847.1 1752.28  5998.3 1758.14  6059.2 1760.82
#Mann= 9 ,-1 , 0
  3276.9     .05       0  4744.9     .12       0  4985.9     .07       0
  5003.9     .12       0  5123.3     .05       0  5456.2     .12       0
    5647     .05       0  5847.1     .12       0  5998.3     .05       0
Bank Sta=4985.9,5003.9
XS Rating Curve= 0 ,0
Exp/Cntr=0.3,0.1

Type RM Length L Ch R = 1 ,34119   ,528,528,528
BEGIN DESCRIPTION:
Lytle Creek 34576.911
END DESCRIPTION:
XS GIS Cut Line= 4
      1601306.45      6823712.44      1602055.32        6823678.
      1602714.32      6823736.57      1603606.94      6823167.05
#Sta/Elev= 30
  4248.5 1762.21  4597.4 1754.82  4617.4 1752.46  4787.6 1747.97  4807.2 1745.26
  4817.7 1743.45  4837.7  1738.8  4867.7 1744.21  4947.8 1745.92  4967.8  1744.8
  4982.5 1738.11  4986.5 1737.05    4988 1736.55  5004.5 1737.05  5017.9 1737.65
  5032.1 1742.56  5053.9 1745.78  5098.2  1740.3  5128.4 1740.24  5165.6 1749.95
  5198.6 1746.56  5249.5 1746.59  5502.8 1751.45  5854.3    1753  5978.7 1748.39
  6176.7 1748.74  6379.7 1748.25  6546.8 1751.78  6703.7 1756.65  6718.6 1757.26
#Mann= 13 ,-1 , 0
  4248.5     .05       0  4807.2     .12       0  4817.7     .05       0
  4982.5     .12       0  4986.5     .07       0  5004.5     .12       0
  5032.1     .05       0  5249.5     .12       0  5502.8     .05       0
  6176.7     .12       0  6379.7     .05       0  6546.8     .12       0
  6703.7     .05       0
Bank Sta=4986.5,5004.5
XS Rating Curve= 0 ,0
Exp/Cntr=0.3,0.1

Type RM Length L Ch R = 1 ,33591   ,561,561,561
BEGIN DESCRIPTION:
Lytle Creek 33980.178
END DESCRIPTION:
XS GIS Cut Line= 3
      1601447.67      6824182.65      1602261.14      6824140.17
      1603683.66      6823127.21
#Sta/Elev= 30
  4192.3  1760.3  4239.7 1761.12  4343.7 1758.73    4490 1756.21  4610.2 1752.29
  4794.8  1750.8  4870.6 1750.34  4930.6 1748.25  4949.1 1744.56  4960.7 1740.04
  5009.5 1734.34    5011 1733.84  5027.5 1734.34  5033.3 1739.04  5039.4 1739.38
    5048  1742.2  5060.7 1744.35  5089.8 1744.37  5175.9 1749.18  5226.3 1750.33
  5727.9 1752.65    5871 1751.28  5965.2  1747.5  6057.4 1748.61  6110.8 1748.34
  6322.5 1747.92  6474.8 1751.35  6582.5 1753.44  6639.3 1755.95  6753.2 1760.95
#Mann= 9 ,-1 , 0
  4192.3     .05       0  4343.7     .12       0  4794.8     .05       0
  5009.5    .035       0  5027.5     .05       0  6110.8     .12       0
  6322.5     .05       0  6474.8     .12       0  6639.3     .05       0
Bank Sta=5009.5,5027.5
XS Rating Curve= 0 ,0
Exp/Cntr=0.3,0.1
