HEC-RAS study Rainy Creek.prj: Rainy Creek Base Level Engineering

--- Rainy Creek.g01 (geometry) --- (continued)

Type RM Length L Ch R = 1 ,73506   ,496,496,496
BEGIN DESCRIPTION:
Rainy Creek 73505.6
END DESCRIPTION:
XS GIS Cut Line= 4
      1617051.49      6824407.98      1617265.01      6824777.73
      1617421.26      6825043.36      1617799.92      6825173.03
#Sta/Elev= 30
  4573.2 1851.58  4590.4 1851.46  4596.3 1850.64  4606.2 1851.21    4758 1847.58
  4772.8 1847.69  4810.1  1845.5  4884.7 1843.43  4890.5 1842.73  4927.8 1841.11
  4942.8 1839.77  4965.1 1834.35  4965.4 1833.46  4965.9 1832.96  4975.8 1832.96
  4976.3 1833.46  4986.7 1834.73  4992.4 1834.27  4997.4 1834.93  5029.6  1835.4
  5035.4 1836.39  5051.1 1837.38  5081.7 1837.01  5285.4 1838.19  5386.3 1840.29
  5395.7 1840.86  5407.4 1840.52    5566 1842.91  5671.7    1846  5708.6 1847.67
#Mann= 3 ,-1 , 0
  4573.2     .05       0  4965.4     .05       0  4976.3     .05       0
Bank Sta=4965.4,4976.3
XS Rating Curve= 0 ,0
Exp/Cntr=0.3,0.1

Type RM Length L Ch R = 1 ,73010   ,501,501,501
BEGIN DESCRIPTION:
Rainy Creek 73009.9
END DESCRIPTION:
XS GIS Cut Line= 3
      1616377.02      6825075.48      1616952.51      6825132.77
        1617989.      6825221.31
#Sta/Elev= 30
  4423.9 1851.62  4482.2  1851.8  4723.4 1850.16  4843.9 1846.75  4874.1 1845.49
  4934.4 1841.15  4944.4 1839.67  4954.5 1839.55  4984.6 1832.18  4989.2  1829.7
  4989.7  1829.2  4999.6  1829.2  5000.1  1829.7    5001 1831.29  5007.4 1831.63
  5014.8 1833.03  5034.8 1832.78    5075 1834.86  5105.1  1834.1  5145.2 1836.18
  5165.3 1836.51  5335.9 1836.14  5354.2 1837.14  5426.3 1838.91  5657.1 1842.43
  5677.2 1843.44  5687.2 1842.84  5817.7 1847.22  5887.9 1848.39  6042.5 1852.64
#Mann= 3 ,-1 , 0
  4423.9     .05       0  4989.2     .05       0  5000.1     .05       0
Bank Sta=4989.2,5000.1
XS Rating Curve= 0 ,0
Exp/Cntr=0.3,0.1

Type RM Length L Ch R = 1 ,72509   ,174,174,174
BEGIN DESCRIPTION:
Rainy Creek 72508.98
END DESCRIPTION:
XS GIS Cut Line= 3
      1616482.57      6825532.85      1617088.01      6825528.51
      1617999.42       6825500.3
#Sta/Elev= 30
  4388.3  1851.3  4600.7 1848.29  4620.7 1845.85  4640.7 1846.41  4650.7 1846.24
  4660.7 1845.31  4710.7 1844.64  4800.7 1839.78  4820.7 1837.64  4860.7 1835.17
  4880.7 1832.17  4890.7 1831.28  4910.7  1831.4  4940.7  1829.8  4945.2 1828.97
  4945.7 1828.47  4955.7 1828.47  4956.2 1828.97  5010.8  1831.7  5070.8 1831.86
  5168.9 1834.28  5180.8 1835.42  5190.8 1835.12  5260.9 1837.13    5471 1839.84
    5531 1841.74    5551 1842.88  5681.1 1846.51  5822.3 1849.77  5905.6 1850.37
#Mann= 3 ,-1 , 0
  4388.3     .05       0  4945.2     .05       0  4956.2     .05       0
Bank Sta=4945.2,4956.2
XS Rating Curve= 0 ,0
Exp/Cntr=0.3,0.1

Type RM Length L Ch R = 1 ,72335   ,643,643,643
BEGIN DESCRIPTION:
Rainy Creek 72334.82
END DESCRIPTION:
XS GIS Cut Line= 3
      1616330.66      6825749.86      1617159.63      6825684.76
      1618101.81      6825665.27
#Sta/Elev= 30
  4168.1 1851.63  4282.8 1851.38    4343 1852.22  4380.8 1849.95  4423.2 1851.95
  4493.4 1851.42  4533.6 1849.95  4553.6 1847.27  4593.7 1847.28  4724.1 1843.12
    4768 1840.85  4834.5 1836.39  4884.6 1830.06  4944.8 1829.96  4959.4 1829.32
  4959.9 1828.82  4969.9 1828.82  4970.4 1829.32  4974.9 1829.86    5035 1829.64
    5045 1829.86    5065 1831.57    5095 1832.56  5455.1 1838.48  5545.1 1841.99
  5564.2 1841.89  5575.1 1842.73  5625.1 1843.71  5745.1 1845.78    5942 1846.59
#Mann= 3 ,-1 , 0
  4168.1     .05       0  4959.4     .03       0  4970.4     .05       0
Bank Sta=4959.4,4970.4
XS Rating Curve= 0 ,0
Exp/Cntr=0.3,0.1

Type RM Length L Ch R = 1 ,71692   ,600,600,600
BEGIN DESCRIPTION:
Rainy Creek 71692.31
END DESCRIPTION:
XS GIS Cut Line= 3
      1616799.37      6826357.51      1617301.99      6826281.99
       1618377.5      6826203.86
#Sta/Elev= 30
  4485.1 1846.53  4515.8 1846.61  4561.6 1845.38  4662.7 1844.23  4844.7 1837.91
  4914.8 1833.95  4919.9 1834.44  4925.6 1833.14    4956 1831.08  4976.2  1825.6
  4986.8 1823.69  4987.3 1823.19  4997.4 1823.19  4997.9 1823.69  5016.4 1826.41
  5056.5 1825.71  5267.1 1830.36  5457.6 1831.77  5547.8 1834.57  5718.3 1838.57
  5728.3 1839.89  5738.3 1839.67  5748.4  1838.2  5758.4 1838.46  5768.4 1839.63
  5848.6 1841.28  5928.8 1843.87  5944.7 1844.88  5949.7 1844.46  6071.7 1847.52
#Mann= 3 ,-1 , 0
  4485.1     .05       0  4986.8     .05       0  4997.9     .05       0
Bank Sta=4986.8,4997.9
XS Rating Curve= 0 ,0
Exp/Cntr=0.3,0.1

Type RM Length L Ch R = 1 ,71092   ,567,567,567
BEGIN DESCRIPTION:
Rainy Creek 71091.68
END DESCRIPTION:
XS GIS Cut Line= 3
      1617005.79      6826574.96      1617552.64      6826741.62
       1617919.8       6827056.7
#Sta/Elev= 30
    4425  1838.8    4588 1833.17  4729.8 1829.16  4762.6 1827.35  4790.1 1824.35
  4873.7 1823.76  4884.2 1823.12  4905.1 1822.93    4926 1823.79    4932  1824.5
  4957.3 1824.89  5002.6 1824.14  5025.5 1822.83    5026 1822.33  5036.3 1822.33
  5036.8 1822.83  5052.5 1824.27  5137.6 1826.14  5201.2  1828.4  5307.7 1834.48
  5350.5 1835.88  5364.7 1837.43  5371.3 1836.58  5421.5 1837.66  5428.4 1837.94
  5442.7 1839.76  5449.3 1837.87  5456.9 1837.69  5463.5 1838.81  5480.5 1839.34
#Mann= 3 ,-1 , 0
    4425     .05       0  5025.5     .05       0  5036.8     .05       0
Bank Sta=5025.5,5036.8
XS Rating Curve= 0 ,0
Exp/Cntr=0.3,0.1

Type RM Length L Ch R = 1 ,70525   ,685,685,685
BEGIN DESCRIPTION:
Rainy Creek 70524.55
END DESCRIPTION:
XS GIS Cut Line= 3
      1616977.31      6826827.11       1617314.1      6827231.61
      1617666.54      6827601.41
#Sta/Elev= 30
  4475.6 1835.15  4645.6 1827.53  4744.5  1824.6  4857.8 1823.64  4929.4  1822.1
  4950.2 1822.13  4964.5 1821.14  4985.3 1821.34  5035.5 1819.62  5049.7 1820.67
  5056.6  1819.8    5099 1819.81    5143  1818.8  5143.5  1818.3  5153.9  1818.3
  5154.4  1818.8  5155.6 1819.88  5169.8 1820.87  5176.7 1823.19  5183.9 1824.18
  5190.9 1825.94  5240.6 1828.83  5275.8 1830.27    5283 1830.08  5289.9 1830.67
  5311.3 1831.02  5318.2  1831.6  5325.5 1831.42  5403.2  1833.6  5512.8 1835.63
#Mann= 3 ,-1 , 0
  4475.6     .05       0    5143     .05       0  5154.4     .05       0
Bank Sta=5143,5154.4
XS Rating Curve= 0 ,0
Exp/Cntr=0.3,0.1

Type RM Length L Ch R = 1 ,69840   ,224,224,224
BEGIN DESCRIPTION:
Rainy Creek 69839.97
END DESCRIPTION:
XS GIS Cut Line= 3
      1616860.97      6826938.16      1616873.13      6827689.94
      1616883.54       6828578.8
#Sta/Elev= 30
  4250.2 1835.16  4380.1 1831.12  4470.1 1827.93  4520.1 1825.42  4590.1  1823.7
  4680.1 1820.33  4790.1 1818.57  4860.1 1818.89  4920.1 1817.44  4930.1 1816.58
  4970.1 1816.85  5010.1 1814.79  5040.1 1815.54  5054.4 1814.69  5054.9 1814.19
  5065.4 1814.19  5065.9 1814.69  5110.1 1816.11  5150.2 1816.17  5190.2 1818.65
  5240.2 1819.55  5250.2 1819.12  5420.2 1819.33  5450.2 1817.42  5460.2 1817.33
  5540.2  1818.6  5570.2 1818.43  5640.2  1820.6  5860.2 1830.58    5891 1831.33
#Mann= 3 ,-1 , 0
  4250.2     .05       0  5054.4     .05       0  5065.9     .05       0
Bank Sta=5054.4,5065.9
XS Rating Curve= 0 ,0
Exp/Cntr=0.3,0.1

Type RM Length L Ch R = 1 ,69616   ,255,255,255
BEGIN DESCRIPTION:
Rainy Creek 69801.739
END DESCRIPTION:
XS GIS Cut Line= 3
      1616668.26      6827242.03      1616664.67      6827737.21
      1616678.68      6828519.79
#Sta/Elev= 30
  4504.8 1833.78  4610.8 1831.01  4650.8 1828.51  4730.8 1825.65  4760.8 1823.43
  4820.8 1820.99  4870.8  1816.6  4900.8 1815.28  4930.8 1815.21  4980.8 1813.96
  5010.8 1813.95  5030.8 1813.11  5040.8 1814.13  5070.8 1814.96  5110.8 1813.99
  5135.1  1812.8  5135.6  1812.3  5146.1  1812.3  5146.6  1812.8  5150.8 1814.31
  5160.8 1816.16  5170.8  1816.5  5460.9 1816.52  5480.9 1815.33  5510.9 1815.55
  5540.9  1816.9  5580.9 1820.24  5620.9 1822.31  5680.9 1826.51  5782.7 1829.36
#Mann= 3 ,-1 , 0
  4504.8     .05       0  5135.1     .05       0  5146.6     .05       0
Bank Sta=5135.1,5146.6
XS Rating Curve= 0 ,0
Exp/Cntr=0.3,0.1

Type RM Length L Ch R = 1 ,69361   ,398,398,398
BEGIN DESCRIPTION:
Rainy Creek 69360.629
END DESCRIPTION:
XS GIS Cut Line= 3
      1616505.01      6827537.98      1616425.09      6827788.23
        1616305.      6828388.02
#Sta/Elev= 30
  4737.3 1826.47  4790.8 1824.61  4817.8 1822.85    4850  1821.7  4855.2 1822.01
  4887.4 1819.69  4894.8 1818.22  4914.3 1816.88  4919.6 1817.15  4946.5 1813.29
  4951.8 1813.67  4957.8 1812.21  4997.3 1811.32  5050.8 1811.79  5085.8 1811.05
  5086.3 1810.55  5096.8 1810.55  5097.3 1811.05  5152.7  1813.3  5162.9 1811.45
  5173.1 1811.32  5203.7 1811.49  5229.5 1812.72  5280.4 1813.93  5285.5 1813.59
  5397.5 1818.07  5438.4 1820.73  5479.1 1822.16  5581.1 1828.56  5611.7 1829.38
#Mann= 3 ,-1 , 0
  4737.3     .05       0  5085.8     .05       0  5097.3     .05       0
Bank Sta=5085.8,5097.3
XS Rating Curve= 0 ,0
Exp/Cntr=0.3,0.1

Type RM Length L Ch R = 1 ,68963   ,657,657,657
BEGIN DESCRIPTION:
Rainy Creek 68884.305
END DESCRIPTION:
XS GIS Cut Line= 3
      1616074.92      6827328.36      1616076.11      6827938.16
      1616085.34      6828359.56
#Sta/Elev= 30
  4390.2 1826.17  4459.8 1822.08  4519.8 1820.42  4539.8 1818.87  4569.8 1818.12
  4589.8 1817.03  4779.8 1813.47  4799.8 1813.39  4819.8 1814.06  4829.8 1813.12
  4919.8 1812.89  4939.8 1811.77  4959.8  1808.9  5039.9 1807.97    5054 1806.96
  5054.5 1806.46  5065.3 1806.46  5065.8 1806.96  5079.9 1810.26  5119.9 1817.49
  5129.9 1818.09  5149.9 1818.82  5176.3 1820.79  5209.9 1822.41  5239.9 1823.12
  5249.9 1823.87  5319.9 1825.82  5359.9 1826.26  5369.9 1827.13  5421.5 1828.29
#Mann= 3 ,-1 , 0
  4390.2     .05       0    5054     .05       0  5065.8     .05       0
Bank Sta=5054,5065.8
XS Rating Curve= 0 ,0
Exp/Cntr=0.3,0.1

Type RM Length L Ch R = 1 ,68306   ,463,463,463
BEGIN DESCRIPTION:
Rainy Creek 68306.08
END DESCRIPTION:
XS GIS Cut Line= 3
      1615642.34      6827244.26      1615551.19      6827686.98
      1615412.29      6828322.88
#Sta/Elev= 30
  4553.6 1823.95    4569 1823.56    4588 1824.33  4598.3 1824.16  4614.2 1823.11
  4649.3 1823.26  4709.7 1822.47  4765.1 1818.68    4782 1817.07  4792.2 1814.24
  4810.4  1811.9  4860.7 1808.77  4884.1 1805.74  4910.2  1803.7  4910.7  1803.2
  4921.6  1803.2  4922.1  1803.7  4945.4 1805.35  4961.3 1805.79  4986.2 1805.41
  5003.6 1804.52  5016.9 1804.57  5060.5 1808.85  5078.3 1809.55  5339.3 1815.58
  5476.1 1819.67  5530.2 1820.69  5579.9  1822.3  5641.3 1823.12  5656.5 1823.96
#Mann= 3 ,-1 , 0
  4553.6     .05       0  4910.2     .05       0  4922.1     .05       0
Bank Sta=4910.2,4922.1
XS Rating Curve= 0 ,0
Exp/Cntr=0.3,0.1

Type RM Length L Ch R = 1 ,67843   ,109,109,109
BEGIN DESCRIPTION:
Rainy Creek 67842.83
END DESCRIPTION:
XS GIS Cut Line= 3
      1615064.51      6827192.96      1615120.06      6827599.17
      1615238.08      6828373.23
#Sta/Elev= 30
  4600.2 1826.67  4605.3 1826.06  4640.7 1825.43  4736.5 1824.88  4756.7  1823.3
  4790.2 1822.19  4817.2 1820.39  4837.4 1821.67  4857.4 1819.73  4867.7 1819.42
    4898 1816.36  4918.2 1811.28  4939.7 1810.66  4958.5 1809.16  4988.8  1802.2
  5104.2 1802.02  5104.7 1801.52  5115.7 1801.52  5116.2 1802.02  5261.9 1802.08
  5276.1 1802.65  5339.6 1808.83  5408.2 1812.08  5476.8 1814.67  5494.6 1814.69
  5514.8 1816.14  5575.5 1818.09  5696.9 1820.61    5741 1822.13  5793.2  1822.4
#Mann= 3 ,-1 , 0
  4600.2     .05       0  5104.2     .05       0  5116.2     .05       0
Bank Sta=5104.2,5116.2
XS Rating Curve= 0 ,0
Exp/Cntr=0.3,0.1

Type RM Length L Ch R = 1 ,67734   ,118,118,118
BEGIN DESCRIPTION:
Rainy Creek 67733.73
END DESCRIPTION:
XS GIS Cut Line= 4
      1614953.39      6827286.66      1615026.31       6827644.3
      1615057.56      6827852.64      1615144.37       6828460.3
#Sta/Elev= 30
  4641.1 1822.49  4777.3 1819.98  4856.8  1814.7  4873.3 1809.66  4901.8 1809.44
  4902.3 1808.94  4913.8 1809.44  4923.8 1814.15  4928.9 1815.23  4938.4 1815.99
  4974.3 1814.09  4979.4 1817.14  5010.5 1817.29    5020 1815.87  5040.2 1817.62
  5161.1 1817.08  5166.2 1815.24  5230.6 1816.69  5235.7 1814.61  5301.3 1816.32
  5306.4  1813.8  5363.6 1815.07  5372.1 1814.51  5377.1 1812.23  5383.8 1811.64
  5434.3 1811.11  5454.5 1811.65  5474.7 1814.92  5525.2 1816.76  5830.6 1821.12
#Mann= 3 ,-1 , 0
  4641.1     .05       0  4901.8     .05       0  4913.8     .05       0
Bank Sta=4901.8,4913.8
XS Rating Curve= 0 ,0
Exp/Cntr=0.3,0.1

Type RM Length L Ch R = 1 ,67616   ,477,477,477
BEGIN DESCRIPTION:
Rainy Creek 67615.91
END DESCRIPTION:
XS GIS Cut Line= 4
      1614817.98      6827272.81      1614908.25       6827644.3
      1614929.09      6827883.89      1614995.06      6828529.74
#Sta/Elev= 30
  4620.5 1821.19  4646.4 1820.47  4677.3 1818.19  4728.7 1815.99  4780.2 1812.94
  4802.2 1812.73  4831.7 1811.27  4885.7 1810.02  4944.9 1807.25  4955.1 1806.58
  4975.7 1801.63    4986 1801.92  4996.1 1801.13  4996.6 1800.63  5007.7 1800.63
  5008.2 1801.13  5027.3 1802.86  5066.7  1802.3  5096.9 1803.23    5127 1803.25
  5177.2 1802.45  5207.3 1804.22  5257.5 1805.88  5446.3 1810.71  5478.6 1812.63
  5619.3  1815.9  5739.6 1816.47  5744.6 1817.31  5770.1 1817.94  5892.5 1817.53
#Mann= 3 ,-1 , 0
  4620.5     .05       0  4996.1     .05       0  5008.2     .05       0
Bank Sta=4996.1,5008.2
XS Rating Curve= 0 ,0
Exp/Cntr=0.3,0.1

Type RM Length L Ch R = 1 ,67139   ,360,360,360
BEGIN DESCRIPTION:
Rainy Creek 67138.96
END DESCRIPTION:
XS GIS Cut Line= 3
       1614292.8      6827403.12      1614516.76      6827879.69
      1614750.58      6828565.55
#Sta/Elev= 30
  4478.3 1814.94  4543.4 1815.35    4550 1814.63  4640.1 1817.62  4708.5 1817.39
  4793.1 1812.81  4837.3 1808.26  4859.4 1803.92  4903.6 1799.26  4964.9  1797.9
  4980.9 1796.77  5001.2 1797.86  5016.9 1797.45  5024.2 1798.74  5055.9 1798.39
  5073.6 1796.72  5074.1 1796.22  5085.7 1796.72  5087.6 1799.25  5105.7 1801.75
    5151 1803.38  5293.7 1805.26  5450.5 1808.57  5476.5 1808.23  5489.1 1809.21
  5570.5 1809.01  5575.8 1809.98  5669.9 1810.72  5721.5 1813.06  5729.5  1812.6
#Mann= 3 ,-1 , 0
  4478.3     .05       0  5073.6     .03       0  5085.7     .05       0
Bank Sta=5073.6,5085.7
XS Rating Curve= 0 ,0
Exp/Cntr=0.3,0.1

Type RM Length L Ch R = 1 ,66779   ,342,342,342
BEGIN DESCRIPTION:
Rainy Creek 66779.21
END DESCRIPTION:
XS GIS Cut Line= 3
      1613725.06      6827512.47      1614209.47      6828041.15
      1614584.03      6828423.51
#Sta/Elev= 30
  4288.3 1818.18  4518.6 1817.69  4589.5 1816.63  4624.7  1817.3  4638.9 1816.18
  4688.8 1814.93  4752.3 1811.41  4787.5    1808  4809.1 1806.96  4815.8 1805.84
  4851.6    1803  4858.4 1801.97  4872.6 1801.69  4879.4 1799.62  4886.8  1798.4
  4907.7 1796.49  4950.3 1795.29  4972.6 1793.96  4973.1 1793.46  4984.2 1793.46
  4984.7 1793.96  5014.2 1794.52  5063.6 1798.55  5091.9 1799.49  5289.9    1802
  5431.4 1805.03  5445.5 1804.77  5473.8  1805.6  5494.9 1805.36  5540.6 1806.09
#Mann= 3 ,-1 , 0
  4288.3     .05       0  4972.6     .05       0  4984.7     .05       0
Bank Sta=4972.6,4984.7
XS Rating Curve= 0 ,0
Exp/Cntr=0.3,0.1

Type RM Length L Ch R = 1 ,66437   ,333,333,333
BEGIN DESCRIPTION:
Rainy Creek 66436.99
END DESCRIPTION:
XS GIS Cut Line= 3
      1613313.65      6828009.91      1613954.26      6828231.25
      1614574.07      6828525.54
#Sta/Elev= 30
  4325.8 1809.14    4521 1810.02    4560 1811.43    4578 1808.52  4602.3 1810.79
  4739.9 1809.36  4765.1 1807.68    4791 1808.58  4835.1 1807.85  4930.3 1802.56
  4940.9 1800.93    4962 1795.08  4972.6 1792.03  4978.1 1788.88  5002.6 1787.54
  5003.1 1787.04  5014.9 1787.54    5026  1788.2  5031.5 1790.57  5048.7 1792.09
  5059.8 1796.16  5082.5 1800.91  5099.7 1802.12  5122.4 1801.38    5128 1798.53
  5137.2 1796.55  5145.2 1796.49  5218.9 1799.02  5474.4 1802.39  5689.7 1807.75
#Mann= 3 ,-1 , 0
  4325.8     .05       0  5002.6     .05       0  5014.9     .05       0
Bank Sta=5002.6,5014.9
XS Rating Curve= 0 ,0
Exp/Cntr=0.3,0.1

Type RM Length L Ch R = 1 ,66104   ,438,438,438
BEGIN DESCRIPTION:
Rainy Creek 66104.13
END DESCRIPTION:
XS GIS Cut Line= 4
      1613178.23      6828267.72      1613764.16      6828483.86
       1613852.7       6828509.9       1614516.8       6828632.3
#Sta/Elev= 30
  4377.2 1804.13  4501.7 1803.89  4512.8 1803.02  4851.4 1799.19  4887.2 1797.91
  4937.4 1797.68  4942.7 1798.61  4967.8 1798.73  4973.2 1799.55  5036.6 1799.82
  5064.7 1799.62    5070 1798.49    5086 1800.06  5097.7 1799.77  5111.4 1795.65
  5116.7 1794.99    5141 1793.49  5141.5 1792.99  5153.3 1793.49    5198 1794.08
  5381.1 1799.38  5492.6 1800.66  5543.8 1802.69  5555.7 1802.16  5584.4 1802.66
  5614.9 1804.62  5635.3  1804.2  5666.8 1804.92  5726.8 1807.87  5769.3  1808.3
#Mann= 3 ,-1 , 0
  4377.2     .05       0    5141     .03       0  5153.3     .05       0
Bank Sta=5141,5153.3
XS Rating Curve= 0 ,0
Exp/Cntr=0.3,0.1

Type RM Length L Ch R = 1 ,65666   ,680,680,680
BEGIN DESCRIPTION:
Rainy Creek 65665.53
END DESCRIPTION:
XS GIS Cut Line= 3
       1612861.3      6828499.86      1613590.43      6828860.95
      1614360.65       6829207.9
#Sta/Elev= 30
  4192.1 1797.62    4307 1798.35  4419.2 1797.66  4542.5 1792.66    4649 1791.11
  4664.9 1791.53  4671.4 1790.89  4865.8 1792.12  4901.3 1790.18  4918.1 1790.22
  4923.7 1789.19  4946.1 1787.74    4963 1789.33  4977.4 1789.41  5037.5 1786.57
    5038 1786.07  5049.8 1786.57  5082.9 1789.49  5088.4 1791.19  5106.1 1792.05
  5111.5 1793.14  5152.3 1794.54  5227.2 1798.71  5250.4 1798.91  5353.9 1803.33
    5614 1809.54  5800.4 1811.56  5822.4 1812.67  5833.2 1811.94  5850.5 1812.38
#Mann= 3 ,-1 , 0
  4192.1     .05       0  5037.5     .05       0  5049.8     .05       0
Bank Sta=5037.5,5049.8
XS Rating Curve= 0 ,0
Exp/Cntr=0.3,0.1

Type RM Length L Ch R = 1 ,64986   ,576,576,576
BEGIN DESCRIPTION:
Rainy Creek 64985.63
END DESCRIPTION:
XS GIS Cut Line= 3
      1612663.34      6828475.53      1612937.65      6828940.81
      1613455.02      6829485.96
#Sta/Elev= 30
  4463.3 1794.86  4538.6 1794.37  4554.2 1793.68  4575.7 1794.18  4591.3 1793.32
  4721.6 1791.46  4751.3 1790.36  4757.1 1790.75  4772.8 1790.18  4794.2 1788.55
  4809.9 1786.49  4831.3 1785.39  4840.8 1782.87  4841.3 1782.37  4852.7 1782.37
  4853.2 1782.87  4884.1 1784.67  4932.8 1785.45  4969.9 1785.42  4985.6 1784.05
  5013.5 1783.62  5027.7 1784.43    5035 1786.16  5077.4 1787.98  5331.9 1795.25
  5339.1 1794.48  5367.5  1794.4  5600.8 1796.66  5629.2 1797.46    5755 1797.97
#Mann= 3 ,-1 , 0
  4463.3     .05       0  4840.8     .05       0  4853.2     .05       0
Bank Sta=4840.8,4853.2
XS Rating Curve= 0 ,0
Exp/Cntr=0.3,0.1

Type RM Length L Ch R = 1 ,64410   ,425,425,425
BEGIN DESCRIPTION:
Rainy Creek 64409.51
END DESCRIPTION:
XS GIS Cut Line= 3
      1611996.66      6828683.85      1612413.34      6829083.17
      1613331.72      6829578.75
#Sta/Elev= 30
  4425.3 1792.83  4490.8 1792.28  4688.7 1792.36  4851.6 1791.02  4858.5 1790.16
  4879.9 1789.59  4907.9 1787.23  4936.2 1782.47  4943.4 1780.67  4972.3 1777.84
  4972.8 1777.34  4984.4 1777.34  4984.9 1777.84    5000 1778.31  5015.7 1780.47
  5060.4 1781.33    5126 1784.01  5153.6 1784.09  5197.5 1785.66  5257.4 1785.33
  5339.3 1786.22  5367.9 1787.37  5413.4 1787.63  5492.9 1789.55  5574.4 1790.42
  5663.4 1792.91    5722 1792.59  5760.1 1793.57  5825.7 1793.68    6046 1795.89
#Mann= 3 ,-1 , 0
  4425.3     .05       0  4972.3     .05       0  4984.9     .05       0
Bank Sta=4972.3,4984.9
XS Rating Curve= 0 ,0
Exp/Cntr=0.3,0.1

Type RM Length L Ch R = 1 ,63985   ,389,389,389
BEGIN DESCRIPTION:
Rainy Creek 63984.92
END DESCRIPTION:
XS GIS Cut Line= 3
      1611743.23        6829045.      1612080.01      6829315.81
      1613128.27      6829753.17
#Sta/Elev= 30
  4569.5 1788.33  4623.1 1788.85  4650.6  1788.1  4786.6 1787.39  4900.2 1785.67
  4978.6 1782.16    4993 1780.01  5001.7 1776.85  5022.4 1775.37  5022.9 1774.87
  5034.5 1774.87    5035 1775.37  5061.2 1775.82  5069.5 1776.76  5074.9 1778.69
  5082.9 1780.31  5098.7  1780.2  5122.5 1781.54  5151.8 1780.57  5321.3 1783.58
  5429.6 1784.31  5488.5 1785.83  5548.8 1785.55  5748.4  1788.1  5825.3 1789.72
  5907.6 1790.06  5960.6 1791.12  5984.5 1792.23  6061.3 1792.08  6137.5 1792.75
#Mann= 3 ,-1 , 0
  4569.5     .05       0  5022.4     .05       0    5035     .05       0
Bank Sta=5022.4,5035
XS Rating Curve= 0 ,0
Exp/Cntr=0.3,0.1

Type RM Length L Ch R = 1 ,63596   ,350,350,350
BEGIN DESCRIPTION:
Rainy Creek 63596.17
END DESCRIPTION:
XS GIS Cut Line= 3
      1611380.92      6829289.37      1611808.47      6829593.22
      1612424.82      6829755.98
#Sta/Elev= 30
  4476.6 1784.13  4556.6 1783.39  4600.9 1783.94  4621.8 1782.67  4628.8 1783.41
  4707.9 1781.41    4874 1780.68  4936.7 1779.06  4945.3 1777.75  4951.4 1778.22
  4960.1 1776.36  4966.2 1776.87  4972.3 1775.58    4981 1775.04  5000.9 1775.25
  5028.6 1776.98  5069.9  1776.6  5111.3 1775.62    5132 1774.51  5135.9 1773.31
  5136.4 1772.81  5148.8 1773.31  5157.4 1775.22    5163 1778.12  5173.4 1779.18
  5225.1 1778.22  5307.8  1779.4  5359.5 1781.53    5525 1783.95  5638.6  1783.8
#Mann= 3 ,-1 , 0
  4476.6     .05       0  5135.9     .05       0  5148.8     .05       0
Bank Sta=5135.9,5148.8
XS Rating Curve= 0 ,0
Exp/Cntr=0.3,0.1

Type RM Length L Ch R = 1 ,63246   ,452,452,452
BEGIN DESCRIPTION:
Rainy Creek 63246.22
END DESCRIPTION:
XS GIS Cut Line= 3
      1610911.12      6829761.22      1611803.05      6829910.96
       1612334.7      6829934.83
#Sta/Elev= 30
  4093.8 1782.37  4138.3 1781.91  4178.9 1780.38  4249.8 1779.97  4310.7 1778.23
  4371.5 1777.75  4604.7 1777.59  4655.4 1778.28  4704.8 1780.14  4736.6 1778.63
  4797.4 1777.28  4898.8 1777.65  4929.2 1776.51  4939.3 1775.18  4952.3 1772.85
  4959.6  1770.9  4963.3  1770.5  4963.8    1770  4975.8    1770  4976.3  1770.5
  5070.2 1771.73  5090.3 1773.53  5100.3 1775.01  5120.3 1776.49  5190.4 1778.54
  5210.4 1780.22  5240.4 1779.99  5310.5 1781.22  5400.6 1782.04  5530.4 1782.39
#Mann= 3 ,-1 , 0
  4093.8     .05       0  4963.3     .05       0  4976.3     .05       0
Bank Sta=4963.3,4976.3
XS Rating Curve= 0 ,0
Exp/Cntr=0.3,0.1

Type RM Length L Ch R = 1 ,62794   ,411,411,411
BEGIN DESCRIPTION:
Rainy Creek 62793.83
END DESCRIPTION:
XS GIS Cut Line= 3
      1610745.77      6830270.94      1611657.21      6830317.82
      1612124.74      6830323.01
#Sta/Elev= 30
  4089.3 1775.85  4126.4 1775.25  4208.7 1774.88    4429 1774.55    4469 1774.78
  4529.1 1774.25  4708.9 1774.81  4839.5 1775.89  4849.5 1774.06  4869.6 1774.26
  4906.4 1771.81  4929.6 1771.76  4979.7 1770.48  4989.7 1769.54  4998.3 1768.05
  5003.2 1767.82  5003.7 1767.32  5015.7 1767.32  5016.2 1767.82  5029.7 1772.27
  5039.7 1774.48  5059.7 1774.88  5119.7 1774.05  5199.7 1774.99  5279.7 1776.69
  5339.8 1777.54  5359.8 1777.31  5399.8 1778.03  5429.8 1777.89  5469.5 1778.33
#Mann= 3 ,-1 , 0
  4089.3     .05       0  5003.2     .03       0  5016.2     .05       0
Bank Sta=5003.2,5016.2
XS Rating Curve= 0 ,0
Exp/Cntr=0.3,0.1

Type RM Length L Ch R = 1 ,62383   ,585,585,585
BEGIN DESCRIPTION:
Rainy Creek 62383.43
END DESCRIPTION:
XS GIS Cut Line= 3
      1610672.84      6830630.32      1611451.49      6830630.32
      1612091.05      6830565.32
#Sta/Elev= 30
  4217.9 1776.87  4370.1 1775.54  4550.1 1774.88  4580.1 1773.53  4680.1 1772.94
  4860.1 1773.24  4940.1 1774.27  4990.1 1774.29  4995.8 1771.27  5000.8 1771.27
  5010.1 1767.42  5020.2 1765.55  5023.7 1765.48  5024.2 1764.98  5036.2 1764.98
  5036.7 1765.48  5040.3 1767.61  5050.3 1770.25  5067.2 1771.26  5080.5 1771.48
  5090.5 1770.56  5100.6 1770.54  5160.9 1771.56  5281.5 1771.44  5341.8 1772.87
  5522.8 1772.93  5552.9    1774    5573 1776.69  5593.1 1777.52  5639.4 1777.98
#Mann= 3 ,-1 , 0
  4217.9     .05       0  5023.7     .05       0  5036.7     .05       0
Bank Sta=5023.7,5036.7
XS Rating Curve= 0 ,0
Exp/Cntr=0.3,0.1

Type RM Length L Ch R = 1 ,61798   ,768,768,768
BEGIN DESCRIPTION:
Rainy Creek 61798.47
END DESCRIPTION:
XS GIS Cut Line= 3
      1610540.01       6830867.3      1611803.05      6830890.74
      1612417.67      6830885.53
#Sta/Elev= 30
  3734.2 1779.12  3769.2 1779.14  3809.2 1778.21  3919.2 1777.09  4179.3 1772.37
  4539.3 1772.39  4577.4 1772.01  4599.3 1771.66  4629.3 1766.82  4642.8 1765.49
  4643.3 1764.99  4655.4 1764.99  4655.9 1765.49  4679.4 1770.56  4699.4 1771.81
  4709.4 1771.76  4719.4 1770.24  4759.4 1770.97  4789.4 1769.88  4879.4 1769.38
  4909.4 1768.09  4979.4 1767.24  4995.9 1765.61  5000.9 1765.61  5029.4 1770.05
  5109.4 1773.66  5219.4 1776.85  5319.4 1776.67  5419.4 1777.71  5612.1 1778.23
#Mann= 3 ,-1 , 0
  3734.2     .05       0  4642.8     .05       0  4655.9     .05       0
Bank Sta=4642.8,4655.9
XS Rating Curve= 0 ,0
Exp/Cntr=0.3,0.1

Type RM Length L Ch R = 1 ,61030   ,613,613,613
BEGIN DESCRIPTION:
Rainy Creek 61030.34
END DESCRIPTION:
XS GIS Cut Line= 3
      1610668.12      6831214.85      1611466.68      6831258.25
      1612369.43      6831184.47
#Sta/Elev= 30
  4190.4 1778.06  4247.4 1776.51  4297.4 1776.07  4397.6 1772.44  4447.7 1771.53
  4627.9 1770.71    4648 1770.05    4688  1770.6    4711 1769.85  4908.3 1768.72
  4918.4 1767.42  4928.4 1767.19  4938.4 1765.65  4951.8 1761.53  4952.3 1761.03
  4964.6 1761.03  4965.1 1761.53  4968.4 1762.93  5018.6 1767.05  5038.6 1767.98
  5059.2 1766.61  5078.8 1768.46  5088.8 1768.67  5098.8 1767.96  5108.9 1768.61
  5175.7 1769.29  5269.4 1769.21    5460 1772.66  5730.9 1775.56  5895.9 1776.34
#Mann= 3 ,-1 , 0
  4190.4     .05       0  4951.8     .05       0  4965.1     .05       0
Bank Sta=4951.8,4965.1
XS Rating Curve= 0 ,0
Exp/Cntr=0.3,0.1

Type RM Length L Ch R = 1 ,60417   ,445,445,445
BEGIN DESCRIPTION:
Rainy Creek 60417.4
END DESCRIPTION:
XS GIS Cut Line= 3
      1609865.15      6831761.73      1611557.83      6831809.47
      1612550.88      6831458.21
#Sta/Elev= 30
  3309.4 1774.62  3349.3  1772.9  3379.3 1772.59  3439.3 1770.57  3479.3 1770.55
  3599.4  1768.7  3719.4 1767.97  4279.6 1768.63  4549.7  1767.9  4689.8 1766.37
  4819.9 1766.59  4859.9 1765.76  4919.9 1766.08  4959.9  1764.4  4973.3 1762.71
  4973.8 1762.21  4986.1 1762.21  4986.6 1762.71  4989.9 1764.62  4998.8 1765.46
  5010.4 1764.99  5031.6  1765.5  5049.8 1763.37    5074 1763.41  5111.6 1765.53
  5148.3 1766.29  5384.5 1767.85  5508.9 1771.03  5784.7 1773.48  6056.1 1775.06
#Mann= 3 ,-1 , 0
  3309.4     .05       0  4973.3     .03       0  4986.6     .05       0
Bank Sta=4973.3,4986.6
XS Rating Curve= 0 ,0
Exp/Cntr=0.3,0.1

Type RM Length L Ch R = 1 ,59972   ,724,724,724
BEGIN DESCRIPTION:
Rainy Creek 59972.28
END DESCRIPTION:
XS GIS Cut Line= 5
      1609849.72       6831824.7      1610774.22      6832215.34
      1610883.59      6832239.16      1611497.07      6832239.16
      1612790.28      6832230.48
#Sta/Elev= 30
  3262.5 1773.81  3300.8 1772.96  3344.2 1770.55  3376.8 1770.43  3420.2 1768.63
  3466.4 1767.78  3590.3 1767.89  3648.6 1767.11  4007.5 1766.25  4409.5 1766.33
  4749.5 1763.86  4839.5 1764.05  4869.5 1764.68  4899.5 1763.99  4929.5 1764.01
  4959.5 1765.37  4969.5 1764.26    4981 1760.34  4981.5 1759.84  4994.5 1759.84
    4995 1760.34  5019.5 1763.46  5059.5 1764.41  5159.5 1765.57  5209.5 1765.19
  5309.5 1765.64  5409.5  1767.2  5749.5 1767.55  6069.5 1771.65  6284.8 1772.58
#Mann= 3 ,-1 , 0
  3262.5     .05       0    4981     .05       0    4995     .05       0
Bank Sta=4981,4995
XS Rating Curve= 0 ,0
Exp/Cntr=0.3,0.1

Type RM Length L Ch R = 1 ,59248   ,501,501,501
BEGIN DESCRIPTION:
Rainy Creek 59248.23
END DESCRIPTION:
XS GIS Cut Line= 3
      1609995.36      6832668.85      1611254.01      6832855.48
      1612287.01      6832916.24
#Sta/Elev= 30
  3726.7 1762.76  4009.4 1763.42  4727.2 1763.19  4888.9 1761.04  4929.3 1762.52
  4949.6 1760.24  4969.8 1760.22  4978.5 1758.16    4983 1756.07  4983.5 1755.57
    4997 1756.07  4997.1 1756.72  5002.1 1756.72  5020.1 1761.69  5060.2  1761.1
  5110.3 1762.73  5200.4 1762.97  5230.5 1761.82  5260.6  1762.6  5280.6 1761.51
  5301.6 1762.08  5310.6 1761.19  5466.9  1761.2  5480.9 1760.54    5531 1762.38
  5661.2 1764.29  5841.6 1768.74  5881.6 1770.59  5921.7 1770.53  6033.9 1772.68
#Mann= 3 ,-1 , 0
  3726.7     .05       0    4983     .05       0    4997     .05       0
Bank Sta=4983,4997
XS Rating Curve= 0 ,0
Exp/Cntr=0.3,0.1

Type RM Length L Ch R = 1 ,58747   ,984,984,984
BEGIN DESCRIPTION:
Rainy Creek 58746.75
END DESCRIPTION:
XS GIS Cut Line= 3
      1609923.91      6832716.04      1611293.07      6833259.12
      1612186.96      6833463.07
#Sta/Elev= 30
  3533.5 1762.01  3620.7  1762.3  3689.3 1761.63  3857.4 1762.78    3922 1762.34
  4018.8 1760.43  4199.8 1760.42  4223.2 1761.03  4352.3 1759.18  4391.5 1759.66
    4559 1758.27  4739.6 1759.15  4799.4 1759.91  4804.7 1760.58  4829.1 1759.81
  4907.4 1760.55    5010 1759.71  5023.8 1756.91    5032 1756.28  5032.5 1755.78
  5045.8 1755.78  5046.3 1756.28    5072 1760.28  5109.8 1763.03  5200.9 1766.54
  5264.8 1767.82    5292 1769.23    5335 1769.36  5340.2 1768.78  5923.3 1774.94
#Mann= 3 ,-1 , 0
  3533.5     .05       0    5032     .05       0  5046.3     .05       0
Bank Sta=5032,5046.3
XS Rating Curve= 0 ,0
Exp/Cntr=0.3,0.1

Type RM Length L Ch R = 1 ,57763   ,888,888,888
BEGIN DESCRIPTION:
Rainy Creek 57763.26
END DESCRIPTION:
XS GIS Cut Line= 3
       1609818.6      6832813.41       1610569.5      6833594.69
      1610950.72      6833845.95
#Sta/Elev= 30
  3924.6 1762.22  4137.6  1759.8  4201.1  1760.7  4278.8 1758.88  4370.9 1758.84
  4455.8 1757.59  4526.6 1757.26  4554.9 1758.04  4590.1 1756.46  4639.5 1756.19
  4759.9 1757.53  4830.7 1757.36    4859 1756.39  4873.1 1754.37    4887  1754.1
  4887.5  1753.6  4901.4  1754.1  4908.4 1756.43  4929.6 1756.82    4986 1755.57
  4993.3 1754.43  5043.1 1754.18  5058.2 1755.28  5064.2 1758.14  5073.3  1758.4
  5079.3 1760.56  5100.3 1762.25  5151.5 1763.84  5238.9 1764.96  5464.8 1765.04
#Mann= 3 ,-1 , 0
  3924.6     .05       0    4887     .05       0  4901.4     .05       0
Bank Sta=4887,4901.4
XS Rating Curve= 0 ,0
Exp/Cntr=0.3,0.1

Type RM Length L Ch R = 1 ,56875   ,793,793,793
BEGIN DESCRIPTION:
Rainy Creek 56875.33
END DESCRIPTION:
XS GIS Cut Line= 4
      1609653.69      6832891.53      1609753.52      6833503.54
      1609905.43      6833941.91       1610382.9      6834093.83
#Sta/Elev= 30
  4386.9 1761.05  4422.4 1760.63    4515 1760.88  4545.3 1760.24  4606.2 1759.91
  4678.4 1760.06  4768.3 1759.25  4808.9 1757.93  4889.9 1756.55  4940.6 1756.06
  4960.9 1756.32    4971 1756.11  4980.6 1754.23  4985.7 1753.93  4994.1 1751.64
  4994.6 1751.14  5008.2 1751.14  5008.7 1751.64    5107 1754.74  5255.1 1754.18
  5426.8 1755.66    5481 1755.24  5554.4  1755.5  5617.4  1756.4  5636.3 1757.14
  5673.8 1757.61  5738.2 1759.64  5743.5 1759.38  5802.7 1760.61    5972 1761.13
#Mann= 3 ,-1 , 0
  4386.9     .05       0  4994.1     .05       0  5008.7     .05       0
Bank Sta=4994.1,5008.7
XS Rating Curve= 0 ,0
Exp/Cntr=0.3,0.1

Type RM Length L Ch R = 1 ,56082   ,584,584,584
BEGIN DESCRIPTION:
Rainy Creek 56082.45
END DESCRIPTION:
XS GIS Cut Line= 4
      1609520.45       6833246.8      1609437.12      6834038.48
      1609681.91      6834163.48      1610286.06      6834121.81
#Sta/Elev= 30
  3930.5 1758.97  3971.9 1758.22  4121.8  1757.5  4213.3 1755.38  4263.5 1755.27
  4303.7  1754.6  4333.9  1755.4  4364.1 1754.27  4464.6 1753.35  4665.7 1753.75
  4827.6 1752.07  4881.4 1752.84  4955.4 1752.38  4971.2 1751.49  4983.2 1748.82
  4986.4 1747.44  4986.9 1746.94  5000.5 1746.94    5001 1747.44  5004.9  1748.6
    5009 1748.09  5014.5 1749.06  5024.6 1752.11  5074.7  1753.7  5114.8 1753.62
    5195 1754.39  5335.3  1754.4  5425.5  1756.4  5455.6 1758.11    5607 1760.03
#Mann= 3 ,-1 , 0
  3930.5     .05       0  4986.4     .05       0    5001     .05       0
Bank Sta=4986.4,5001
XS Rating Curve= 0 ,0
Exp/Cntr=0.3,0.1

Type RM Length L Ch R = 1 ,55498   ,1689,1689,1689
BEGIN DESCRIPTION:
Rainy Creek 55112.27
END DESCRIPTION:
XS GIS Cut Line= 3
      1608029.36      6835460.54       1609702.8      6834431.92
      1611453.87      6833720.93
#Sta/Elev= 30
  3035.7 1773.71  3064.6 1772.92  3085.8 1768.48  3107.1 1766.59  3339.1 1758.47
  3412.5  1759.9  3623.2 1756.91  3665.7 1754.74    3864  1754.8  4145.7 1751.13
  4380.5 1750.58  4707.4 1751.91  4771.2  1753.3    4918 1750.51  4945.2  1747.9
  4954.7 1750.17  4960.6 1748.97  4967.4 1750.19  4981.9 1749.81    5000 1747.97
  5021.1  1749.3  5026.5 1747.07  5037.9 1746.91  5038.4 1746.41  5052.6 1746.91
  5080.1 1747.84  5110.3 1752.27    5313 1752.64    5771 1761.09  6889.9 1767.97
#Mann= 3 ,-1 , 0
  3035.7     .05       0  5037.9     .05       0  5052.6     .05       0
Bank Sta=5037.9,5052.6
XS Rating Curve= 0 ,0
Exp/Cntr=0.3,0.1

Type RM Length L Ch R = 1 ,53809   ,642,642,642
BEGIN DESCRIPTION:
Rainy Creek 54125.452
END DESCRIPTION:
XS GIS Cut Line= 3
      1608305.04      6835937.98      1609405.33      6835446.42
      1610717.78      6834097.99
#Sta/Elev= 30
  3794.9 1800.29  3855.6 1799.83    3902 1795.34  3907.5 1792.83  3925.3 1793.32
  3930.7 1790.48  3953.9 1789.52  3959.4  1786.7  3977.1 1785.13  3982.6 1781.59
  4000.4 1780.84  4005.8 1777.88  4052.3 1770.83  4057.7 1768.24  4248.9 1755.43
  4370.4 1753.14  4520.6 1754.36  4830.3 1749.05  4876.5 1748.69  4944.9 1749.34
  4960.3 1747.98  4968.9    1742  4969.4  1741.5  4986.6    1742  4997.1 1745.06
  5076.5 1748.02  5203.8 1746.25  6214.9 1751.79  6674.6 1761.32  6881.7 1762.78
#Mann= 5 ,-1 , 0
  3794.9     .05       0  4830.3     .12       0  4876.5     .05       0
  4968.9     .05       0  4986.6     .05       0
Bank Sta=4968.9,4986.6
XS Rating Curve= 0 ,0
Exp/Cntr=0.3,0.1

Type RM Length L Ch R = 1 ,53167   ,640,640,640
BEGIN DESCRIPTION:
Rainy Creek 53167.01
END DESCRIPTION:
XS GIS Cut Line= 4
      1607997.52      6836394.15      1609407.28      6836088.59
      1609747.56      6835975.74      1611540.04      6836236.15
#Sta/Elev= 30
  3554.2 1797.44  3715.3 1797.22  3807.4 1794.29  3892.2  1785.3  3941.4 1777.08
  3980.4 1765.36  4022.3 1764.36  4042.8 1767.54  4078.8 1764.98  4083.9 1767.09
  4114.4 1766.46  4196.3    1758  4298.6  1756.2  4441.8 1758.43  4462.3  1756.2
  4544.1 1757.18  4666.9 1751.63  4972.3 1746.44  5008.6 1740.78  5009.1 1740.28
  5026.4 1740.78  5036.4 1745.41    5044 1745.71    5472 1746.52  5635.6 1744.71
  5726.5 1747.78  5746.7 1743.21    5777 1747.23  6605.6 1750.05  7166.5 1759.21
#Mann= 3 ,-1 , 0
  3554.2     .05       0  5008.6     .05       0  5026.4     .05       0
Bank Sta=5008.6,5026.4
XS Rating Curve= 0 ,0
Exp/Cntr=0.3,0.1

Type RM Length L Ch R = 1 ,52527   ,781,781,781
BEGIN DESCRIPTION:
Rainy Creek 52526.88
END DESCRIPTION:
XS GIS Cut Line= 4
      1607858.65      6837151.09        1609567.      6836664.98
       1609833.3      6836539.98       1611170.6      6836357.76
#Sta/Elev= 30
  3212.6 1793.08  3364.8 1790.83  3389.5 1788.37  3423.4 1779.69  3489.5 1772.22
  3520.7 1764.77  3681.2 1758.23  3687.1 1756.14  3884.6 1752.27  3905.4 1757.49
  3978.2 1756.79  4084.9 1754.56  4165.3  1749.5  4196.9  1752.4  4331.7 1754.33
  4488.6 1752.42  4945.1    1745  4960.1 1744.29  4976.2 1739.14  4976.7 1738.64
  4994.1 1739.14  5008.7 1742.67  5038.4 1743.85  5345.2  1744.4  5456.2  1743.4
  5476.4 1740.29  5506.7 1745.46  5526.9 1745.79  6122.3 1746.55  6632.6 1752.75
#Mann= 3 ,-1 , 0
  3212.6     .05       0  4976.2     .05       0  4994.1     .05       0
Bank Sta=4976.2,4994.1
XS Rating Curve= 0 ,0
Exp/Cntr=0.3,0.1

Type RM Length L Ch R = 1 ,51746   ,632,632,632
BEGIN DESCRIPTION:
Rainy Creek 51745.57
END DESCRIPTION:
XS GIS Cut Line= 4
      1608132.68      6837633.65      1610129.24       6837069.4
      1610554.59      6836743.88      1611460.84      6836470.71
#Sta/Elev= 30
  2919.9 1784.34    2998 1786.93  3071.2 1784.27  3105.1 1773.68  3110.3 1775.29
  3130.1 1764.21  3161.3 1755.58  3212.3 1748.79  3275.6 1752.29  3363.7 1750.68
  3452.3 1745.08  3483.5 1749.44  3549.2 1749.28    3577 1745.98  3639.3 1747.28
  3734.6 1741.89  3768.6 1744.45  4578.4 1741.05  4949.3 1742.71    4978    1742
  4994.7 1739.18  4996.1 1736.21  4996.6 1735.71  5017.2 1736.21  5027.5 1740.17
  5056.6 1738.88  5071.1 1742.46  5249.7 1741.26  5697.8 1745.87  6476.8 1758.37
#Mann= 3 ,-1 , 0
  2919.9     .05       0  4996.1     .05       0  5017.2     .05       0
Bank Sta=4996.1,5017.2
XS Rating Curve= 0 ,0
Exp/Cntr=0.3,0.1

Type RM Length L Ch R = 1 ,51114   ,1732,1732,1732
BEGIN DESCRIPTION:
Rainy Creek 51114.02
END DESCRIPTION:
XS GIS Cut Line= 4
      1607946.85      6837847.47      1610299.24      6837543.65
      1610875.62      6837543.66       1611650.8      6837345.96
#Sta/Elev= 30
  2630.4 1786.21  2664.5 1778.28  2669.6 1780.25  2709.2 1772.05  2738.9  1761.7
  2743.9 1762.88  2769.7 1758.45  2880.6 1759.48  2920.9 1754.44  3011.7 1751.38
  3041.9 1754.47  3072.2 1750.06  3122.6 1752.96  3203.3 1751.15    3415 1741.18
  3586.4 1739.02  4147.3 1738.52  4877.1  1740.2  4937.6 1739.62  4941.7 1736.13
  4942.2 1735.63  4973.8 1736.13  5002.3 1736.62  5058.1  1743.3  5582.3  1745.4
    5618 1738.84    5640 1742.16  5781.5 1741.63  6042.5 1750.65  6378.7 1756.02
#Mann= 3 ,-1 , 0
  2630.4     .05       0  4941.7     .05       0  4973.8     .05       0
Bank Sta=4941.7,4973.8
XS Rating Curve= 0 ,0
Exp/Cntr=0.3,0.1

Type RM Length L Ch R = 1 ,49382   ,1251,1251,1251
BEGIN DESCRIPTION:
Rainy Creek 49382.17
END DESCRIPTION:
XS GIS Cut Line= 3
      1607794.88      6838142.61      1608801.84      6838242.44
      1611550.91      6838611.24
#Sta/Elev= 30
  3988.5 1789.06  4119.3 1787.16  4139.4 1783.03  4194.9 1764.23  4199.9 1768.49
  4219.7 1762.65  4259.9 1759.34    4280 1759.84  4300.9  1754.8  4360.4 1751.29
  4521.2 1745.81  4598.6 1751.42  4631.8 1751.27  4704.6  1747.9  4742.3 1743.64
  4812.6 1742.69  4832.7 1740.14    4883 1743.68  4901.4 1739.23  4906.4 1740.04
  4923.2 1737.01  4967.3 1735.33  4967.9 1734.83  4999.6 1735.33  5002.5 1737.24
  5225.4 1736.72  5518.2 1739.51  5861.2 1736.46  6661.3 1744.75  7774.1 1749.02
#Mann= 3 ,-1 , 0
  3988.5     .05       0  4967.3     .05       0  4999.6     .05       0
Bank Sta=4967.3,4999.6
XS Rating Curve= 0 ,0
Exp/Cntr=0.3,0.1

Type RM Length L Ch R = 1 ,48131   ,725,725,725
BEGIN DESCRIPTION:
Rainy Creek 48131.19
END DESCRIPTION:
XS GIS Cut Line= 3
      1608063.99      6838915.18      1609461.56      6839088.79
      1610850.24      6839379.54
#Sta/Elev= 30
  3597.8 1785.65  3810.4 1785.88  3921.3 1784.92  3931.4 1783.91  3981.2 1766.53
  3986.2 1765.82  3991.8 1762.57  4001.9 1759.07  4032.1 1752.19  4082.5  1746.7
  4183.3 1740.85  4223.6 1739.39  4253.8 1739.83  4324.4  1737.6  4435.2 1736.22
  4596.4 1735.76  4719.1 1736.63  4818.1 1734.53  4918.9 1734.84  5010.4 1733.06
  5014.7 1731.17  5015.3 1730.67  5047.1 1731.17  5050.5 1734.11  5060.7 1735.13
  5125.7 1734.54  5183.3 1736.28    5515 1737.85  5999.1 1744.16  6424.9 1748.03
#Mann= 3 ,-1 , 0
  3597.8     .05       0  5014.7     .05       0  5047.1     .05       0
Bank Sta=5014.7,5047.1
XS Rating Curve= 0 ,0
Exp/Cntr=0.3,0.1

Type RM Length L Ch R = 1 ,47406   ,212,212,212
BEGIN DESCRIPTION:
Rainy Creek 47405.64
END DESCRIPTION:
XS GIS Cut Line= 3
      1608239.22      6839675.16      1609253.14      6839741.13
      1610777.46      6839734.19
#Sta/Elev= 30
  3981.6 1782.01  4047.5 1783.31  4217.9 1782.03  4237.9 1777.66  4247.9  1774.3
  4254.7 1770.32  4259.7 1771.07    4298 1758.68  4358.2 1745.69  4378.2  1743.8
  4438.3 1742.02  4478.4 1744.73  4518.5 1738.13  4528.5 1737.54  4638.8 1735.78
  4688.9 1736.92    4739 1734.59  4879.3 1733.81  4929.4 1732.05  4939.4 1733.19
  4979.8 1730.43  4980.4 1729.93  5012.3 1730.43  5029.5 1735.94  5039.5 1737.68
  5059.5 1733.78  5089.5 1733.01  5369.5 1735.46  5839.5 1736.76    6522 1748.19
#Mann= 3 ,-1 , 0
  3981.6     .05       0  4979.8     .03       0  5012.3     .05       0
Bank Sta=4979.8,5012.3
XS Rating Curve= 0 ,0
Exp/Cntr=0.3,0.1

Type RM Length L Ch R = 1 ,47194   ,597,597,597
BEGIN DESCRIPTION:
Rainy Creek 47193.8
END DESCRIPTION:
XS GIS Cut Line= 3
      1608360.74        6839946.      1609253.14      6839952.94
      1610720.94      6839966.82
#Sta/Elev= 30
    4106  1781.1  4140.3 1780.86  4190.3 1777.77  4240.3 1768.61  4250.3 1765.88
  4270.3 1757.81  4280.3 1755.39  4320.3 1750.07  4390.3 1743.19  4480.3 1742.96
  4660.3  1738.3  4880.3  1734.5  4910.3 1732.97  4950.3 1733.18  4960.3 1731.82
    4964 1728.71  4964.6 1728.21  4996.5 1728.71  4996.9 1730.39  5020.3 1729.65
  5060.3 1732.76  5200.3 1733.58  5250.3 1732.69  5300.3 1734.35  5350.3 1734.61
  5810.3 1734.96  5990.3 1736.46  6120.3 1738.86  6220.3  1742.4  6466.3 1747.84
#Mann= 3 ,-1 , 0
    4106     .05       0    4964     .03       0  4996.5     .05       0
Bank Sta=4964,4996.5
XS Rating Curve= 0 ,0
Exp/Cntr=0.3,0.1

Type RM Length L Ch R = 1 ,46597   ,523,523,523
BEGIN DESCRIPTION:
Rainy Creek 46597.3
END DESCRIPTION:
XS GIS Cut Line= 3
      1608264.91      6840189.05      1609556.62      6840381.76
      1610831.35      6840329.73
#Sta/Elev= 30
  3695.5 1772.69  3715.8 1769.52    3736 1761.37  3756.3 1760.62  3766.4 1757.35
  3806.8 1750.49    3827 1750.69    3918  1744.9  3948.4  1744.7  3978.7 1749.82
    4009 1745.34  4057.8 1746.34  4170.8 1744.41  4251.7  1742.1  4271.9 1740.01
  4504.4 1734.97    4879 1732.31  4959.4 1728.18  4979.6 1729.16  4993.6 1726.61
  4994.2 1726.11  5026.1 1726.61  5029.9  1730.3  5049.9 1732.81    5150 1729.52
    5180 1732.86  5210.1 1733.77  5480.3 1733.27  5750.5 1735.28  6277.3 1748.89
#Mann= 3 ,-1 , 0
  3695.5     .05       0  4993.6     .05       0  5026.1     .05       0
Bank Sta=4993.6,5026.1
XS Rating Curve= 0 ,0
Exp/Cntr=0.3,0.1

Type RM Length L Ch R = 1 ,46074   ,856,856,856
BEGIN DESCRIPTION:
Rainy Creek 46073.55
END DESCRIPTION:
XS GIS Cut Line= 3
      1608509.71      6841038.02      1609535.78      6840834.88
      1611050.68      6840449.65
#Sta/Elev= 30
  3940.8 1737.74  4139.9 1738.63  4327.8 1737.96  4532.7 1735.21  4896.4 1732.83
  4947.7 1731.44  4975.8 1726.76  4983.8 1726.46  5006.6 1727.61  5027.3 1727.36
  5047.9 1729.08  5058.2 1728.73  5058.3 1725.98  5058.9 1725.48  5090.9 1725.98
  5099.5 1730.44  5120.7 1731.02  5161.6 1731.25    5182 1727.63  5197.4 1726.25
  5243.9 1730.99  5264.6 1730.05  5279.3 1731.13  5367.8 1732.67    5636 1732.41
  5806.1 1734.52  5969.8 1738.28  6110.7 1743.68  6275.8  1747.8  6549.9 1752.56
#Mann= 3 ,-1 , 0
  3940.8     .05       0  5058.3     .05       0  5090.9     .05       0
Bank Sta=5058.3,5090.9
XS Rating Curve= 0 ,0
Exp/Cntr=0.3,0.1

Type RM Length L Ch R = 1 ,45218   ,406,406,406
BEGIN DESCRIPTION:
Rainy Creek 45217.58
END DESCRIPTION:
XS GIS Cut Line= 3
      1608619.11      6841386.97      1609895.16      6841428.63
      1611176.41      6841433.84
#Sta/Elev= 30
  3713.9 1736.84  3779.8 1737.49  3889.9 1736.77    4010 1734.46    4050 1734.46
    4070  1733.5  4290.1 1729.49  4370.1    1729  4490.2 1729.76  4508.4 1729.04
  4540.2 1729.89  4710.3 1730.38  4830.4 1729.56  4920.4 1726.49  4970.5 1727.56
  4993.1 1726.46    5004 1725.02  5004.6 1724.52    5037 1725.02  5050.5 1727.93
  5060.5 1729.07  5110.5 1727.91  5150.5 1728.63  5180.5 1727.33  5200.5 1728.55
  5310.5 1729.88  5720.5 1738.24  5930.5 1741.53    6065 1746.06  6271.9 1749.84
#Mann= 3 ,-1 , 0
  3713.9     .05       0    5004     .05       0    5037     .05       0
Bank Sta=5004,5037
XS Rating Curve= 0 ,0
Exp/Cntr=0.3,0.1

Type RM Length L Ch R = 1 ,44812   ,519,519,519
BEGIN DESCRIPTION:
Rainy Creek 44811.67
END DESCRIPTION:
XS GIS Cut Line= 3
      1608671.18      6841803.63      1609806.62      6841803.63
      1610874.31      6841855.72
#Sta/Elev= 30
  3865.9 1736.76  4139.7 1735.78  4149.7 1734.19  4229.7  1733.7  4239.7 1730.71
  4259.7 1729.43  4299.7  1728.3  4469.7 1727.81  4539.7 1728.42  4959.7 1729.06
  4989.7 1727.04  4993.2  1721.6  4993.8  1721.1  5025.7  1721.1  5026.3  1721.6
  5029.8 1725.04  5059.8 1725.37  5069.8 1723.85  5079.8 1725.49  5089.8 1726.11
  5149.9 1727.64    5230 1727.55  5350.1 1730.77  5380.2 1730.91  5490.3 1735.45
  5760.6 1743.68  5780.6 1745.19  5840.7  1745.3  5910.8 1747.66  6070.3 1749.45
#Mann= 3 ,-1 , 0
  3865.9     .05       0  4993.2     .05       0  5026.3     .05       0
Bank Sta=4993.2,5026.3
XS Rating Curve= 0 ,0
Exp/Cntr=0.3,0.1

Type RM Length L Ch R = 1 ,44293   ,515,515,515
BEGIN DESCRIPTION:
Rainy Creek 44292.51
END DESCRIPTION:
XS GIS Cut Line= 3
      1608748.87      6842198.84      1609755.84      6842307.35
      1610337.42      6842572.09
#Sta/Elev= 30
  3987.9 1732.87    4125 1731.64  4315.9 1726.79  4436.6 1725.74  4798.7 1727.12
    4859  1725.1  4929.4 1725.18  4939.5 1727.38  4949.6 1727.69  4979.7 1726.61
  4997.8 1721.66  5009.8 1720.94  5021.7 1722.59  5032.7 1726.42  5038.4 1730.21
  5054.7  1731.9  5065.7 1725.14  5076.7 1719.13    5137 1718.66  5137.6 1718.16
  5170.1 1718.66  5175.6 1718.66  5187.7 1725.96  5197.5 1728.06  5210.7 1728.66
  5228.3  1734.9  5251.3 1732.57  5264.2 1733.11  5582.1 1743.68  5639.7 1744.35
#Mann= 5 ,-1 , 0
  3987.9     .05       0  5065.7     .12       0    5137     .03       0
  5170.1     .12       0  5264.2     .05       0
Bank Sta=5137,5170.1
XS Rating Curve= 0 ,0
Exp/Cntr=0.3,0.1

Type RM Length L Ch R = 1 ,43778   ,618,618,618
BEGIN DESCRIPTION:
Rainy Creek 43778.37
END DESCRIPTION:
XS GIS Cut Line= 3
      1608818.36      6842424.54      1609547.51      6842754.39
      1610010.98      6843109.58
#Sta/Elev= 30
  4207.5 1728.62  4275.8 1728.78  4327.5 1726.87  4357.5 1728.69  4425.5 1728.37
  4523.4 1724.13    4662 1725.26  4904.1 1724.31  4972.1 1725.54  4994.1    1725
  5006.1 1721.64  5022.7 1723.48  5029.8 1721.34  5072.6 1725.73  5122.4 1720.12
    5137 1724.21  5151.5 1725.41  5157.8 1721.91    5166  1723.2  5170.2 1718.26
  5170.8 1717.76  5203.4 1718.26  5236.7 1719.91  5251.2 1725.99    5272 1730.39
  5301.1  1729.7  5336.4 1732.34  5350.9 1731.77  5550.3 1740.45  5591.7 1740.02
#Mann= 3 ,-1 , 0
  4207.5     .05       0  5170.2     .03       0  5203.4     .05       0
Bank Sta=5170.2,5203.4
XS Rating Curve= 0 ,0
Exp/Cntr=0.3,0.1

Type RM Length L Ch R = 1 ,43160   ,633,633,633
BEGIN DESCRIPTION:
Rainy Creek 43160.02
END DESCRIPTION:
XS GIS Cut Line= 4
      1608750.77      6842394.97      1608798.47      6842593.53
       1609191.6      6843210.12       1609495.4      6843691.87
#Sta/Elev= 30
  4069.8 1729.47    4235 1725.91    4463 1725.23  4499.4  1724.2  4535.8 1721.79
  4578.1 1724.03    4760 1723.97  4832.8 1724.72    4854 1723.62  4926.8 1722.85
    4942 1720.38  4946.6  1718.8  4947.2  1718.3  4979.2  1718.3  4979.8  1718.8
  4984.3 1720.05  4999.5 1720.28  5020.7 1722.06  5026.7 1723.48    5036 1723.65
  5041.9 1725.52    5050 1722.56    5109 1722.67  5193.8 1725.75  5203.1 1725.39
  5345.6 1731.04  5404.7 1731.35  5418.6 1732.09  5485.6 1731.47  5574.8 1732.56
#Mann= 3 ,-1 , 0
  4069.8     .05       0  4946.6     .05       0  4979.8     .05       0
Bank Sta=4946.6,4979.8
XS Rating Curve= 0 ,0
Exp/Cntr=0.3,0.1

Type RM Length L Ch R = 1 ,42527   ,586,586,586
BEGIN DESCRIPTION:
Rainy Creek 42526.6
END DESCRIPTION:
XS GIS Cut Line= 4
      1608667.45      6842308.25      1608677.95      6842533.91
      1608753.23      6843592.07      1608787.87      6844284.77
#Sta/Elev= 30
  3725.8 1731.53  3775.6 1731.12  3805.6 1730.22  3825.7 1730.61  3845.7 1729.02
  3895.7 1726.46    4016 1724.69  4497.2 1722.92  4567.3 1721.87  4607.4 1719.87
  4637.5 1720.28  4667.6  1722.1  4697.7 1722.11  4727.7 1722.92  4807.9 1721.74
  4829.5 1722.14    4848 1720.78  4868.1 1721.29  4948.3 1720.07  4970.2 1719.04
  4971.8 1716.16  4972.4 1715.66  5004.4 1715.66    5005 1716.16    5008 1723.34
  5068.5 1724.01  5108.6    1726  5168.7 1726.36  5228.7 1727.85  5706.1    1728
#Mann= 3 ,-1 , 0
  3725.8     .05       0  4971.8     .05       0    5005     .05       0
Bank Sta=4971.8,5005
XS Rating Curve= 0 ,0
Exp/Cntr=0.3,0.1

Type RM Length L Ch R = 1 ,41941   ,812,812,812
BEGIN DESCRIPTION:
Rainy Creek 41941.41
END DESCRIPTION:
XS GIS Cut Line= 3
      1608588.31      6842038.24      1608236.74      6843392.41
      1607972.47      6844414.84
#Sta/Elev= 30
  3620.5 1734.19  3695.5 1732.74  3736.1 1732.94  3852.6 1729.74  3868.2 1728.42
    4096 1723.56  4457.1  1721.8  4486.1 1722.53  4591.4 1721.36  4653.5 1722.09
  4688.9 1720.88  4810.6 1721.31  4901.4 1719.28    4984 1720.93  4994.3 1719.25
  5003.1 1716.27  5008.2 1715.57  5008.7 1714.65  5009.3 1714.15    5042 1714.65
  5048.8 1718.42  5056.3 1721.02  5118.3 1721.22    5139 1720.27  5211.4 1721.46
  5287.5  1723.4  5335.2 1725.83  5376.5 1726.31  5683.5 1726.19  6075.6 1724.41
#Mann= 3 ,-1 , 0
  3620.5     .05       0  5008.7     .05       0    5042     .05       0
Bank Sta=5008.7,5042
XS Rating Curve= 0 ,0
Exp/Cntr=0.3,0.1

Type RM Length L Ch R = 1 ,41129   ,1027,1027,1027
BEGIN DESCRIPTION:
Rainy Creek 41128.53
END DESCRIPTION:
XS GIS Cut Line= 5
      1608449.42      6841877.65      1607733.27       6842884.6
      1607646.46      6843192.76      1607585.32      6843660.36
      1607617.15       6843891.5
#Sta/Elev= 30
  3455.4 1734.69    3559 1732.31  3731.2 1726.61    4046 1721.91    4548 1720.44
  4902.4 1720.74  4960.4 1719.81  4975.1  1716.4  4977.8 1712.94  4978.4 1712.44
  5011.1 1712.94  5011.2 1716.87  5016.5    1718  5036.7 1719.02  5056.4 1718.97
    5077 1715.16  5087.1 1714.25  5117.3 1714.33  5157.7 1716.24  5177.8 1719.31
  5208.1 1720.38  5214.2 1721.54  5278.7 1722.61  5298.9 1724.07  5450.9 1725.62
  5516.4 1725.01  5530.9 1725.83  5588.4 1724.64  5682.3 1724.68  5716.1 1723.87
#Mann= 3 ,-1 , 0
  3455.4     .05       0  4977.8     .03       0  5011.1     .05       0
Bank Sta=4977.8,5011.1
XS Rating Curve= 0 ,0
Exp/Cntr=0.3,0.1
