--- T1 to Elm Creek.prj (project) ---

Proj Title=Tributary No. 1 to Elm Creek Base Level Engineering
Current Plan=p01
Default Exp/Contr=0.3,0.1
English Units
Geom File=g01
Flow File=f01
Plan File=p01
Y Axis Title=Elevation
X Axis Title(PF)=Main Channel Distance
X Axis Title(XS)=Station
BEGIN DESCRIPTION:
Tributary No. 1 to Elm Creek
END DESCRIPTION:
DSS Export Rating Curves= 0
DSS Export Rating Curve Sorted= 0
DSS Export Volume Flow Curves= 0
DXF OffsetX= 0
DXF OffsetY= 0
DXF ScaleX= 1
DXF ScaleY= 10

--- T1 to Elm Creek.p01 (plan) ---

Plan Title=Multiple Run
Program Version=4.10
Short Identifier=Multiple
Geom File=g01
Flow File=f01
Subcritical Flow
K Sum by GR= 0
Std Step Tol= 0.01
Critical Tol= 0.01
Num of Std Step Trials= 20
Max Error Tol= 0.3
Flow Tol Ratio= 0.001
Split Flow NTrial= 30
Split Flow Tol= 0.02
Split Flow Ratio= 0.02
Log Output Level= 0
Friction Slope Method= 1
Unsteady Friction Slope Method= 2
Unsteady Bridges Friction Slope Method= 1
Parabolic Critical Depth
Global Vel Dist= 1 , 1 , 1
Global Log Level= 0
CheckData=True
Encroach Param=-1 ,0,0, 0
BEGIN DESCRIPTION:
Multiple Run
END DESCRIPTION:
Computation Interval=1HOUR
Output Interval=1HOUR
Run HTab= 0
Run UNet= 0
Run PostProcess= 0
Run WQNet= 0
UNET Theta= 1
UNET Theta Warmup= 1
UNET ZTol= 0.02
UNET ZSATol= 0.05
UNET MxIter= 20
UNET MaxInSteps= 0
UNET DtIC= 0
UNET DtMin= 0
UNET MaxCRTS= 20
UNET WFStab= 2
UNET SFStab= 1
UNET WFX= 1
UNET SFX= 1
UNET DSS MLevel= 4
UNET DZMax Abort= 100
UNET Convert EG Bridges= 0
UNET Use Existing IB Tables=-1
UNET Froude Reduction=False
UNET Froude Limit= 1
UNET Froude Power= 10
UNET Time Slicing=0,0, 5
UNET Junction Losses=0
Instantaneous Interval=1HOUR
Write IC File= 0
Write IC File at Sim End=0
Echo Input=False
Echo Parameters=False
Echo Output=False
Write Detailed= 0
WQ AD Non Conservative
WQ ULTIMATE=-1
WQ Max Comp Step=1HOUR
WQ Output Interval=15MIN
WQ Output Selected Increments= 0
WQ Output face flow=0
WQ Output face velocity=0
WQ Output face area=0
WQ Output face dispersion=0
WQ Output cell volume=0
WQ Output cell surface area=0
WQ Output cell continuity=0
WQ Output cumulative cell continuity=0
WQ Output face conc=0
WQ Output face dconc_dx=0
WQ Output face courant=0
WQ Output face peclet=0
WQ Output face adv mass=0
WQ Output face disp mass=0
WQ Output cell mass=0
WQ Output cell source sink temp=0
WQ Output cell source sink nsm=0
WQ Output MaxMinRange=-1
WQ Daily Max Min Mean=-1
WQ Daily Range=0
WQ Daily Time=0
WQ Create Restart=0
WQ Fixed Restart=0
WQ System Summary=0
WQ Use Fixed Temperature=0
Sorting and Armoring Iterations= 10
XS Update Threshold= 0.02
Hydraulics Update Threshold= 0.02
Energy Slope Method= 1
Volume Change Method= 0
XS Weighting Method= 0
Number of US Weighted Cross Sections= 1
Number of DS Weighted Cross Sections= 1
Upstream XS Weight=0.25
Main XS Weight=0.5
Downstream XS Weight=0.25
Number of DS XS's Weighted with US Boundary= 1
Upstream Boundary Weight= 1
Weight of XSs Associated with US Boundary= 0
Number of US XS's Weighted with DS Boundary= 1
Downstream Boundary Weight= 0.5
Weight of XSs Associated with DS Boundary= 0.5
Sediment Output Level= 4
Mass or Volume Output= 0
Output Increment Type= 1
Profile and TS Output Increment= 10
XS Output Flag= 0
XS Output Increment= 10
Disregard all LS=0
Disregard all Conn=0
Disregard all Breaches=0
Disregard all Pumps=0

--- T1 to Elm Creek.f01 (steady flow) ---

Flow Title=Multiple
Number of Profiles=7
Profile Names=10-year,25-year,50-year,1pct_min,100-year,1pct_plu,500-year
River Rch & RM= Tributary No. 1 ,Reach-1,34134
     282     388     474     288     574    1145     853
River Rch & RM= Tributary No. 1 ,Reach-1,23487
     457     642     796     489     976    1948    1491
River Rch & RM= Tributary No. 1 ,Reach-1,14267
     496     698     865     532    1062    2119    1622
River Rch & RM= Tributary No. 1 ,Reach-1,6939
     539     760     944     581    1159    2313    1776
Boundary for River Rch & Prof#=Tributary No. 1 ,Reach-1,1
Up Type=0
Dn Type=3
Dn Slope=0.005
Boundary for River Rch & Prof#=Tributary No. 1 ,Reach-1,2
Up Type=0
Dn Type=3
Dn Slope=0.005
Boundary for River Rch & Prof#=Tributary No. 1 ,Reach-1,3
Up Type=0
Dn Type=3
Dn Slope=0.005
Boundary for River Rch & Prof#=Tributary No. 1 ,Reach-1,4
Up Type=0
Dn Type=3
Dn Slope=0.005
Boundary for River Rch & Prof#=Tributary No. 1 ,Reach-1,5
Up Type=0
Dn Type=3
Dn Slope=0.005
Boundary for River Rch & Prof#=Tributary No. 1 ,Reach-1,6
Up Type=0
Dn Type=3
Dn Slope=0.005
Boundary for River Rch & Prof#=Tributary No. 1 ,Reach-1,7
Up Type=0
Dn Type=3
Dn Slope=0.005

--- T1 to Elm Creek.g01 (geometry) ---

Geom Title=Existing Conditions

River Reach=Tributary No. 1 ,Reach-1
Reach XY= 30
      1556455.00      6814338.00      1557007.90      6816680.08
      1557699.17      6817435.70      1558365.94      6819248.02
      1558797.42      6819334.65      1558105.63      6820128.29
      1558803.84      6821347.44      1558613.02      6822541.31
      1559153.61      6822999.48      1559008.08      6823480.32
      1559649.95      6823835.72      1559818.23      6824701.81
      1560498.88      6825529.92      1562285.62      6825917.35
      1562213.02      6826494.34      1563541.63      6827374.22
      1564041.32      6828774.74      1564404.99      6828395.07
      1564766.35      6828836.65      1565399.82      6828843.44
      1565291.36      6829675.06      1565911.76      6829597.12
      1566606.03      6830334.54      1567179.41      6829960.68
      1567563.14      6831244.06      1569394.52      6832528.20
      1569009.96      6833290.53      1569688.55      6833520.86
      1569912.73      6834594.50      1570905.00      6835388.00

Type RM Length L Ch R = 1,34134,267,267,267
BEGIN DESCRIPTION:
Tributary No. 1 to Elm Creek 39.0
END DESCRIPTION:
XS GIS Cut Line= 3
      1556629.76      6817292.64      1557138.76      6817106.12
      1557980.21      6816257.60
#Sta/Elev= 30
  4150.9 1850.96  4242.0 1849.53  4273.6 1847.44  4284.3 1848.92  4297.7 1848.34
  4305.6 1846.53  4353.4 1845.59  4378.6 1844.02  4401.4 1845.72  4409.1 1844.26
  4422.7 1843.45  4531.1 1842.89  4710.2 1839.72  4752.7 1840.04  4766.8 1838.89
  4872.9 1840.85  4901.2 1840.54  4908.2 1839.66  4943.6 1840.37  4987.7 1838.00
  4997.8 1837.54  4998.1 1837.04  5002.3 1837.54  5007.2 1840.12  5283.0 1839.07
  5648.9 1843.43  5714.3 1844.49  5763.8 1847.00  5849.2 1847.74  5888.0 1848.90
#Mann=6,-1,0
  4150.9    0.07       0  4987.7   0.035       0  4997.8   0.035       0
  5002.3   0.035       0  5648.9    0.07       0  5849.2   0.035       0
Bank Sta=4997.8,5002.3
Exp/Cntr=0.3,0.1

Type RM Length L Ch R = 1,33867,406,406,406
BEGIN DESCRIPTION:
Tributary No. 1 to Elm Creek 38.0
END DESCRIPTION:
XS GIS Cut Line= 3
      1556668.12      6817541.51      1557473.50      6817081.10
      1558254.95      6816788.02
#Sta/Elev= 30
  4127.8 1848.26  4158.8 1847.29  4164.8 1848.40  4186.4 1848.75  4202.2 1846.91
  4267.0 1846.34  4282.9 1845.36  4310.2 1845.71  4326.0 1844.27  4354.6 1845.74
  4385.1 1843.46  4493.0 1842.86  4567.9 1840.93  4852.9 1838.60  4942.0 1839.05
  4997.8 1836.97  4998.1 1836.47  5002.3 1836.97  5008.4 1838.79  5161.3 1838.23
  5174.6 1837.39  5196.9 1839.13  5215.6 1838.52  5270.7 1838.02  5475.0 1840.62
  5516.3 1842.62  5615.6 1844.17  5697.9 1846.79  5754.9 1849.63  5890.1 1856.84
#Mann=7,-1,0
  4127.8    0.07       0  4997.8    0.07       0  5002.3    0.07       0
  5215.6   0.035       0  5475.0    0.07       0  5615.6   0.035       0
  5754.9    0.07       0
Bank Sta=4997.8,5002.3
Exp/Cntr=0.3,0.1

Type RM Length L Ch R = 1,33461,469,469,469
BEGIN DESCRIPTION:
Tributary No. 1 to Elm Creek 37.0
END DESCRIPTION:
XS GIS Cut Line= 3
      1556798.93      6817657.58      1557681.99      6817414.53
      1558396.05      6817055.58
#Sta/Elev= 30
  4084.1 1845.02  4103.7 1844.38  4121.5 1845.38  4143.2 1843.19  4235.6 1842.98
  4251.6 1841.89  4432.7 1839.55  4692.0 1839.13  4909.8 1837.18  4961.6 1837.72
  4992.7 1836.72  4997.6 1835.57  4998.0 1835.07  5002.4 1835.57  5006.2 1836.79
  5028.5 1836.52  5036.9 1837.42  5081.7 1835.58  5104.1 1835.83  5112.2 1836.99
  5117.8 1836.33  5126.5 1837.76  5140.1 1837.14  5156.9 1837.92  5223.8 1837.65
  5357.8 1841.72  5430.4 1842.28  5519.7 1845.07  5625.7 1849.76  5799.2 1853.68
#Mann=3,-1,0
  4084.1    0.07       0  4997.6    0.07       0  5002.4    0.07       0
Bank Sta=4997.6,5002.4
Exp/Cntr=0.3,0.1

Type RM Length L Ch R = 1,32992,951,951,951
BEGIN DESCRIPTION:
Tributary No. 1 to Elm Creek 36.0
END DESCRIPTION:
XS GIS Cut Line= 3
      1556733.38      6818053.18      1557704.99      6817830.09
      1558454.97      6817488.02
#Sta/Elev= 30
  4003.1 1845.26  4025.3 1844.92  4049.8 1845.96  4056.1 1844.56  4117.6 1843.04
  4148.4 1843.07  4199.7 1841.03  4360.1 1839.16  4815.3 1836.68  4846.1 1837.38
  4959.0 1835.29  4979.5 1832.90  4990.9 1835.08  4997.4 1835.23  4997.6 1832.90
  4997.9 1832.40  5002.1 1832.40  5002.5 1832.90  5002.8 1835.23  5076.9 1835.88
  5085.9 1837.10  5098.9 1836.01  5175.9 1835.66  5424.9 1839.23  5551.1 1842.74
  5582.5 1844.33  5648.8 1845.69  5717.9 1848.01  5735.5 1849.40  5824.3 1850.98
#Mann=3,-1,0
  4003.1    0.07       0  4997.6    0.07       0  5002.5    0.07       0
Bank Sta=4997.6,5002.5
Exp/Cntr=0.3,0.1

Type RM Length L Ch R = 1,32041,489,489,489
BEGIN DESCRIPTION:
Tributary No. 1 to Elm Creek 35.0
END DESCRIPTION:
XS GIS Cut Line= 3
      1557062.59      6818519.95      1558149.15      6818485.71
      1558655.02      6818087.98
#Sta/Elev= 30
  3912.9 1838.89  4132.0 1836.54  4535.6 1835.14  4675.7 1834.13  4769.6 1834.75
  4785.7 1834.17  4855.8 1833.97  4875.8 1833.18  4945.8 1833.37  4955.8 1833.18
  4965.8 1832.07  4985.8 1833.48  4995.4 1833.56  4997.4 1832.07  4997.8 1831.57
  5002.2 1831.57  5002.6 1832.07  5002.7 1833.26  5102.1 1833.58  5151.9 1835.14
  5265.7 1837.22  5294.6 1838.59  5344.3 1839.47  5443.8 1842.38  5458.2 1843.32
  5516.0 1844.63  5551.3 1846.29  5557.6 1845.92  5572.1 1847.14  5643.5 1849.31
#Mann=3,-1,0
  3912.9    0.07       0  4997.4    0.07       0  5002.6    0.07       0
Bank Sta=4997.4,5002.6
Exp/Cntr=0.3,0.1

Type RM Length L Ch R = 1,31552,1148,1148,1148
BEGIN DESCRIPTION:
Tributary No. 1 to Elm Creek 34.0
END DESCRIPTION:
XS GIS Cut Line= 3
      1557245.04      6818995.51      1558366.28      6818884.35
      1558960.81      6818558.74
#Sta/Elev= 30
  3929.8 1837.33  4291.5 1832.99  4412.1 1833.70  4593.0 1832.19  4743.7 1832.58
  4767.5 1831.86  4783.9 1829.91  4804.0 1831.28  4974.9 1831.16  4995.0 1830.30
  4997.4 1828.32  4997.8 1827.82  5002.6 1828.32  5015.1 1828.84  5025.1 1830.74
  5089.3 1832.26  5112.1 1836.07  5119.8 1838.91  5134.9 1839.32  5157.7 1838.48
  5163.4 1836.35  5169.1 1836.33  5179.5 1833.91  5185.2 1834.30  5191.9 1831.72
  5201.3 1830.74  5245.0 1830.60  5288.6 1833.88  5568.1 1838.93  5734.4 1844.52
#Mann=3,-1,0
  3929.8    0.07       0  4997.4    0.07       0  5002.6    0.07       0
Bank Sta=4997.4,5002.6
Exp/Cntr=0.3,0.1

Type RM Length L Ch R = 1,30404,1037,1037,1037
BEGIN DESCRIPTION:
Tributary No. 1 to Elm Creek 33.5
END DESCRIPTION:
XS GIS Cut Line= 3
      1557146.77      6819592.38      1558971.33      6819319.96
      1559176.71      6818825.61
#Sta/Elev= 30
  3333.8 1835.92  3382.6 1834.14  3423.0 1835.04  3483.7 1833.54  3536.0 1834.17
  3600.2 1832.62  3776.9 1831.45  4120.7 1830.78  4171.2 1829.59  4272.3 1829.65
  4302.7 1828.43  4353.2 1829.48  4454.3 1829.42  4494.8 1830.35  4504.9 1829.67
  4687.9 1830.23  4717.2 1830.01  4737.4 1828.93  4752.1 1829.52  4816.3 1828.42
  4919.4 1828.36  4980.1 1827.43  4997.4 1826.16  4997.8 1825.66  5002.6 1826.16
  5019.0 1830.83  5024.1 1830.92  5071.1 1830.18  5299.8 1831.46  5713.9 1837.17
#Mann=3,-1,0
  3333.8    0.07       0  4997.4    0.07       0  5002.6    0.07       0
Bank Sta=4997.4,5002.6
Exp/Cntr=0.3,0.1

Type RM Length L Ch R = 1,29367,1028,1028,1028
BEGIN DESCRIPTION:
Tributary No. 1 to Elm Creek 33.2
END DESCRIPTION:
XS GIS Cut Line= 3
      1557081.38      6819994.90      1558905.88      6819722.48
      1559423.43      6819279.61
#Sta/Elev= 30
  3710.5 1834.60  3805.2 1833.48  3865.8 1834.27  3936.6 1832.20  4191.4 1830.60
  4354.9 1829.87  4563.5 1829.70  4601.3 1828.07  4836.5 1827.67  4937.4 1824.45
  4957.8 1826.73  4978.0 1824.23  4997.4 1823.46  4997.8 1822.96  5002.7 1823.46
  5006.6 1825.74  5080.9 1826.40  5119.6 1826.14  5139.8 1823.46  5150.2 1825.47
  5170.1 1825.55  5190.3 1824.04  5230.8 1826.89  5283.6 1828.40  5291.5 1829.62
  5352.9 1828.28  5422.9 1829.29  5951.5 1829.84  6048.6 1830.29  6236.4 1830.19
#Mann=7,-1,0
  3710.5    0.07       0  4191.4   0.035       0  4354.9    0.07       0
  4997.4    0.07       0  5002.7    0.07       0  5951.5   0.045       0
  6048.6    0.07       0
Bank Sta=4997.4,5002.7
Exp/Cntr=0.3,0.1

Type RM Length L Ch R = 1,28339,728,728,728
BEGIN DESCRIPTION:
Tributary No. 1 to Elm Creek 33.0
END DESCRIPTION:
XS GIS Cut Line= 3
      1557188.50      6820568.38      1558544.30      6820412.70
      1559910.98      6819336.58
#Sta/Elev= 30
  3875.5 1834.07  3902.2 1834.60  4153.8 1830.16  4264.5 1829.14  4314.9 1829.80
  4405.5 1827.39  4475.9 1829.39  4546.4 1827.03  4757.8 1826.47  4818.1 1825.20
  4959.1 1825.23  4989.3 1824.30  4997.3 1820.95  4997.8 1820.45  5002.7 1820.95
  5009.4 1822.48  5019.5 1821.38  5029.5 1824.85  5039.6 1823.63  5130.2 1823.23
  5160.4 1820.95  5180.5 1824.83  5190.6 1825.38  5386.3 1827.31  5508.3 1826.60
  5611.4 1827.67  5655.9 1827.63  6093.1 1828.06  6346.2 1828.35  6979.7 1829.07
#Mann=7,-1,0
  3875.5    0.07       0  4997.3    0.07       0  5002.7    0.07       0
  5611.4   0.045       0  5655.9    0.07       0  6093.1   0.045       0
  6346.2    0.07       0
Bank Sta=4997.3,5002.7
Exp/Cntr=0.3,0.1

Type RM Length L Ch R = 1,27611,435,435,435
BEGIN DESCRIPTION:
Tributary No. 1 to Elm Creek 32.2
END DESCRIPTION:
XS GIS Cut Line= 3
      1557182.56      6821025.56      1559033.80      6821009.06
      1559930.83      6820893.95
#Sta/Elev= 30
  3777.6 1830.39  3900.0 1830.17  3930.0 1830.84  3950.0 1829.74  4040.1 1828.70
  4059.8 1829.33  4100.1 1829.18  4180.1 1827.29  4590.1 1825.54  4670.1 1823.93
  4820.1 1823.21  4860.1 1822.30  4930.1 1821.98  4970.1 1822.64  4980.1 1821.82
  4990.1 1819.69  4997.2 1819.69  4997.7 1819.19  5002.4 1819.19  5002.8 1819.69
  5030.1 1821.91  5100.1 1822.31  5185.8 1821.13  5240.1 1822.89  5424.0 1823.24
  5460.1 1823.91  5532.4 1823.22  5791.4 1823.18  6069.0 1824.55  6533.3 1824.14
#Mann=5,-1,0
  3777.6    0.07       0  4997.2    0.07       0  5002.8    0.07       0
  5424.0   0.035       0  5532.4   0.045       0
Bank Sta=4997.2,5002.8
Exp/Cntr=0.3,0.1

Type RM Length L Ch R = 1,27176,618,618,618
BEGIN DESCRIPTION:
Tributary No. 1 to Elm Creek 32.0
END DESCRIPTION:
XS GIS Cut Line= 3
      1557144.77      6821289.22      1558995.99      6821272.71
      1559891.85      6821157.75
#Sta/Elev= 30
  3437.3 1827.48  4369.1 1823.67  4375.0 1823.68  4597.6 1823.87  4687.6 1822.80
  4877.6 1822.28  4887.6 1821.20  4907.6 1822.27  4977.6 1821.65  4987.6 1821.49
  4997.2 1817.26  4997.7 1816.76  5002.8 1817.26  5007.6 1820.91  5027.6 1817.53
  5037.6 1817.26  5047.6 1820.67  5057.6 1821.20  5087.6 1819.72  5097.6 1818.13
  5127.6 1820.87  5167.6 1821.39  5499.3 1821.98  5518.2 1822.19  5539.6 1823.74
  5620.3 1822.89  5872.4 1824.66  5916.3 1823.88  6084.1 1824.92  6191.8 1824.70
#Mann=5,-1,0
  3437.3    0.07       0  4369.1   0.035       0  4375.0    0.07       0
  4997.2    0.07       0  5002.8    0.07       0
Bank Sta=4997.2,5002.8
Exp/Cntr=0.3,0.1

Type RM Length L Ch R = 1,26558,851,851,851
BEGIN DESCRIPTION:
Tributary No. 1 to Elm Creek 31.5
END DESCRIPTION:
XS GIS Cut Line= 3
      1557170.31      6821912.21      1559055.87      6821826.02
      1559859.49      6821234.12
#Sta/Elev= 30
  3364.8 1825.89  3820.0 1822.33  3940.1 1822.47  3970.1 1821.64  4110.3 1820.78
  4460.6 1820.99  4760.9 1819.31  4821.0 1820.72  4831.0 1820.03  4871.1 1820.13
  4878.3 1819.24  4991.2 1819.48  4997.2 1816.14  4997.7 1815.64  5002.8 1816.14
  5011.2 1816.14  5031.2 1819.02  5061.3 1819.82  5071.3 1821.99  5081.3 1821.69
  5097.9 1819.49  5111.3 1819.75  5131.3 1818.86  5191.4 1819.77  5363.9 1819.79
  5378.6 1820.49  5464.2 1820.68  5487.2 1821.51  5714.8 1822.59  6250.4 1823.10
#Mann=3,-1,0
  3364.8    0.07       0  4997.2    0.07       0  5002.8    0.07       0
Bank Sta=4997.2,5002.8
Exp/Cntr=0.3,0.1

Type RM Length L Ch R = 1,25707,1157,1157,1157
BEGIN DESCRIPTION:
Tributary No. 1 to Elm Creek 31.0
END DESCRIPTION:
XS GIS Cut Line= 3
      1557276.05      6822831.99      1559106.10      6822545.66
      1559788.51      6821664.40
#Sta/Elev= 30
  3604.4 1822.57  4038.6 1822.34  4378.1 1820.69  4463.7 1821.06  4554.8 1819.39
  4666.1 1819.63  4718.6 1818.61  4777.4 1818.13  4825.0 1819.65  4848.3 1818.33
  4909.0 1817.53  4979.9 1817.65  4990.0 1816.37  4997.0 1812.34  4997.5 1811.84
  5003.0 1812.34  5030.5 1817.37  5192.4 1816.60  5216.5 1813.01  5222.8 1813.31
  5232.9 1816.16  5243.0 1816.48  5313.9 1815.89  5341.9 1812.34  5354.4 1815.41
  5384.7 1817.31  5504.3 1817.60  5525.9 1816.78  5996.7 1820.59  6571.3 1821.94
#Mann=5,-1,0
  3604.4    0.07       0  4378.1   0.035       0  4718.6    0.07       0
  4997.0    0.07       0  5003.0    0.07       0
Bank Sta=4997,5003
Exp/Cntr=0.3,0.1

Type RM Length L Ch R = 1,24550,1063,1063,1063
BEGIN DESCRIPTION:
Tributary No. 1 to Elm Creek 30.0
END DESCRIPTION:
XS GIS Cut Line= 3
      1557128.65      6823720.35      1558918.74      6823067.46
      1560219.96      6821388.88
#Sta/Elev= 30
  3046.1 1820.00  3597.0 1819.06  3702.2 1816.04  3769.7 1818.39  3931.7 1818.09
  3994.0 1817.96  4176.2 1816.41  4394.0 1817.04  4613.3 1814.96  4951.5 1815.57
  4956.1 1814.67  4976.2 1811.49  4996.9 1810.74  4997.4 1810.24  5003.1 1810.74
  5005.2 1813.94  5031.4 1814.24  5063.1 1814.42  5077.4 1811.88  5083.9 1812.10
  5090.3 1813.90  5133.7 1811.81  5154.5 1812.75  5177.2 1815.94  5569.2 1816.88
  5812.2 1819.05  6120.5 1820.56  6425.8 1821.14  6447.7 1821.04  7075.4 1821.97
#Mann=11,-1,0
  3046.1    0.07       0  3931.7   0.035       0  3994.0    0.07       0
  4956.1    0.16       0  4996.9    0.07       0  5003.1    0.16       0
  5031.4    0.07       0  5812.2   0.045       0  6120.5    0.07       0
  6425.8   0.045       0  6447.7    0.07       0
Bank Sta=4996.9,5003.1
Exp/Cntr=0.3,0.1

Type RM Length L Ch R = 1,23487,767,767,767
BEGIN DESCRIPTION:
Tributary No. 1 to Elm Creek 29.0
END DESCRIPTION:
XS GIS Cut Line= 3
      1557654.99      6825138.01      1559260.76      6823596.25
      1560414.35      6822356.01
#Sta/Elev= 30
  2773.9 1827.16  3580.1 1816.87  4202.4 1813.64  4379.5 1813.50  4407.8 1815.48
  4443.0 1812.02  4485.5 1812.93  4492.7 1815.35  4513.8 1817.17  4556.2 1811.55
  4744.0 1812.94  4872.5 1812.78  4959.4 1812.67  4996.9 1809.95  4997.4 1809.45
  5003.2 1809.95  5030.0 1813.19  5214.1 1813.56  5331.3 1814.38  5428.6 1814.88
  5531.2 1815.28  5599.2 1815.51  5755.2 1816.31  5792.1 1816.30  5898.9 1816.67
  6037.4 1817.12  6142.8 1817.57  6274.3 1817.77  6429.1 1817.77  6693.8 1818.15
#Mann=17,-1,0
  2773.9    0.07       0  4744.0   0.035       0  4872.5    0.16       0
  4996.9    0.07       0  5003.2    0.16       0  5214.1   0.045       0
  5331.3    0.07       0  5428.6   0.045       0  5531.2    0.07       0
  5599.2   0.045       0  5755.2    0.07       0  5792.1   0.045       0
  5898.9    0.07       0  6037.4   0.045       0  6142.8    0.07       0
  6274.3   0.045       0  6429.1    0.07       0
Bank Sta=4996.9,5003.2
Exp/Cntr=0.3,0.1

Type RM Length L Ch R = 1,22720,656,656,656
BEGIN DESCRIPTION:
Tributary No. 1 to Elm Creek 28.0
END DESCRIPTION:
XS GIS Cut Line= 3
      1558054.98      6825238.01      1559670.14      6823930.63
      1560465.88      6822771.93
#Sta/Elev= 30
  3079.2 1823.06  3619.6 1817.26  4107.0 1814.66  4159.3 1814.95  4214.7 1814.17
  4611.0 1812.11  4835.4 1810.22  4864.2 1808.19  4885.0 1810.14  4956.9 1810.86
  4970.4 1808.43  4992.1 1809.58  4996.8 1807.69  4997.3 1807.19  5003.2 1807.69
  5006.5 1810.12  5086.2 1810.91  5120.0 1808.00  5140.8 1808.75  5155.2 1814.17
  5173.7 1813.91  5191.5 1809.68  5227.3 1807.69  5257.1 1808.56  5284.2 1813.73
  5314.0 1811.37  5384.3 1812.39  6167.4 1816.26  6245.4 1816.11  6562.8 1816.50
#Mann=12,-1,0
  3079.2    0.07       0  4107.0   0.045       0  4159.3    0.07       0
  4214.7   0.045       0  4611.0    0.07       0  4996.8    0.07       0
  5003.2    0.07       0  5086.2    0.16       0  5173.7    0.07       0
  5384.3   0.045       0  6167.4    0.07       0  6245.4   0.045       0
Bank Sta=4996.8,5003.2
Exp/Cntr=0.3,0.1

Type RM Length L Ch R = 1,22064,1008,1008,1008
BEGIN DESCRIPTION:
Tributary No. 1 to Elm Creek 27.0
END DESCRIPTION:
XS GIS Cut Line= 3
      1558485.28      6825503.85      1559905.33      6824405.54
      1560522.45      6823476.68
#Sta/Elev= 30
  3392.9 1820.45  3771.0 1816.57  4058.8 1814.63  4197.7 1813.73  4772.1 1811.10
  4943.6 1808.51  4993.9 1809.56  4995.2 1806.52  4995.7 1806.02  5004.8 1806.52
  5008.4 1808.26  5022.9 1806.52  5036.0 1808.75  5079.1 1809.74  5287.1 1809.56
  5323.1 1807.07  5389.3 1809.59  5446.4 1808.40  5467.5 1809.23  5473.5 1811.55
  5482.5 1811.83  5488.5 1809.48  5518.6 1809.16  5569.4 1810.54  5626.8 1810.04
  5662.9 1812.28  5677.4 1810.49  5699.0 1811.73  5853.6 1812.27  6303.3 1813.62
#Mann=8,-1,0
  3392.9    0.07       0  3771.0   0.045       0  4058.8    0.07       0
  4197.7   0.045       0  4943.6    0.07       0  4995.2    0.07       0
  5004.8    0.07       0  5853.6   0.045       0
Bank Sta=4995.2,5004.8
Exp/Cntr=0.3,0.1

Type RM Length L Ch R = 1,21056,498,498,498
BEGIN DESCRIPTION:
Tributary No. 1 to Elm Creek 26.0
END DESCRIPTION:
XS GIS Cut Line= 3
      1558754.98      6825988.01      1560353.95      6825048.43
      1562155.01      6823037.99
#Sta/Elev= 30
  3145.4 1821.88  3372.0 1817.09  3757.4 1813.56  4600.4 1807.54  4768.6 1806.36
  4956.1 1806.83  4978.0 1804.18  4987.4 1808.09  4993.2 1808.61  4995.2 1804.18
  4995.7 1803.68  5004.9 1804.18  5008.2 1806.44  5029.1 1805.49  5114.2 1806.27
  5192.1 1805.62  5574.9 1809.63  6157.7 1809.67  6208.3 1809.67  6272.3 1809.87
  6360.6 1809.70  6410.3 1811.38  6431.6 1810.24  6990.3 1812.23  7026.7 1811.68
  7033.4 1813.05  7047.6 1813.25  7068.6 1812.08  7211.2 1812.83  7699.2 1818.91
#Mann=11,-1,0
  3145.4    0.07       0  3757.4   0.045       0  4600.4    0.07       0
  4995.2    0.07       0  5004.9    0.07       0  5114.2   0.045       0
  6157.7    0.07       0  6208.3   0.045       0  6272.3    0.07       0
  6990.3   0.035       0  7211.2    0.07       0
Bank Sta=4995.2,5004.9
Exp/Cntr=0.3,0.1

Type RM Length L Ch R = 1,20558,476,476,476
BEGIN DESCRIPTION:
Tributary No. 1 to Elm Creek 25.0
END DESCRIPTION:
XS GIS Cut Line= 3
      1558855.00      6825988.00      1560456.84      6825494.28
      1562454.96      6823888.03
#Sta/Elev= 30
  3323.8 1820.25  3606.3 1814.99  3960.3 1812.28  4477.1 1809.14  4590.0 1809.01
  4820.2 1804.58  4841.1 1806.21  4905.8 1804.32  4924.8 1806.24  4938.5 1804.56
  4987.6 1804.35  4995.1 1800.24  4995.6 1799.74  5004.9 1800.24  5017.4 1804.37
  5102.9 1804.65  5507.2 1803.99  5738.9 1806.32  6070.2 1808.01  6838.2 1807.24
  6880.7 1810.18  6909.4 1800.98  6931.0 1800.26  6945.4 1802.56  6966.2 1808.95
  7051.0 1807.83  7286.2 1814.00  7401.5 1816.64  7506.9 1820.33  7563.7 1819.45
#Mann=11,-1,0
  3323.8    0.07       0  3960.3   0.045       0  4477.1    0.07       0
  4995.1    0.07       0  5004.9    0.07       0  5102.9   0.045       0
  5507.2    0.07       0  5738.9   0.045       0  6880.7    0.07       0
  7286.2   0.035       0  7401.5    0.07       0
Bank Sta=4995.1,5004.9
Exp/Cntr=0.3,0.1

Type RM Length L Ch R = 1,20082,482,482,482
BEGIN DESCRIPTION:
Tributary No. 1 to Elm Creek 24.0
END DESCRIPTION:
XS GIS Cut Line= 3
      1558905.03      6827137.98      1560918.82      6825537.55
      1562455.03      6823937.97
#Sta/Elev= 30
  2427.7 1824.17  2513.4 1824.49  2534.2 1822.37  2675.4 1818.68  3174.6 1812.11
  3790.1 1809.56  3972.8 1808.15  4036.8 1809.65  4078.5 1807.88  4442.1 1806.35
  4484.2 1803.94  4535.1 1806.37  4555.9 1804.44  4812.2 1804.99  4890.7 1808.72
  4897.1 1805.93  4911.5 1804.69  4982.3 1804.50  4995.1 1802.43  4995.6 1801.93
  5004.9 1802.43  5076.4 1802.73  5605.3 1807.14  6480.8 1806.81  6574.2 1809.41
  6616.6 1807.24  6736.8 1807.99  7042.4 1816.21  7129.8 1818.65  7217.8 1819.57
#Mann=10,-1,0
  2427.7   0.035       0  2675.4    0.07       0  3174.6   0.045       0
  3790.1    0.07       0  4995.1    0.07       0  5004.9    0.07       0
  5076.4   0.045       0  6480.8    0.07       0  7042.4   0.035       0
  7129.8    0.07       0
Bank Sta=4995.1,5004.9
Exp/Cntr=0.3,0.1

Type RM Length L Ch R = 1,19600,463,463,463
BEGIN DESCRIPTION:
Tributary No. 1 to Elm Creek 23.0
END DESCRIPTION:
XS GIS Cut Line= 3
      1559305.01      6827387.99      1561307.17      6825794.14
      1562504.98      6823988.03
#Sta/Elev= 30
  2440.9 1821.78  2606.4 1817.14  2669.1 1815.26  2718.8 1803.23  2733.2 1803.26
  2739.6 1808.49  2747.6 1808.38  2754.0 1813.11  2768.4 1813.12  2774.8 1817.96
  2803.7 1823.58  2818.1 1822.32  2838.9 1814.87  2853.3 1813.27  2925.4 1811.05
  3604.5 1808.15  4287.7 1805.19  4419.7 1805.04  4575.4 1801.00  4632.7 1803.71
  4924.8 1802.30  4995.0 1801.00  4995.5 1800.50  5005.0 1801.00  5103.4 1803.38
  5847.3 1806.35  6230.6 1805.09  6663.3 1807.94  7001.3 1817.81  7167.2 1818.86
#Mann=9,-1,0
  2440.9   0.035       0  2606.4    0.07       0  3604.5   0.045       0
  4287.7    0.07       0  4924.8   0.045       0  4995.0   0.045       0
  5005.0   0.045       0  6230.6    0.07       0  7001.3   0.035       0
Bank Sta=4995,5005
Exp/Cntr=0.3,0.1

Type RM Length L Ch R = 1,19137,526,526,526
BEGIN DESCRIPTION:
Tributary No. 1 to Elm Creek 22.0
END DESCRIPTION:
XS GIS Cut Line= 3
      1559755.02      6827887.98      1561740.64      6825888.23
      1562405.02      6824287.96
#Sta/Elev= 30
  2181.9 1816.52  2279.9 1816.78  2397.4 1813.93  2440.4 1813.19  2677.3 1809.57
  2976.7 1807.99  3508.8 1805.48  3836.3 1804.05  4030.7 1803.20  4656.8 1799.27
  4706.2 1802.74  4861.8 1799.29  4946.7 1799.63  4967.9 1802.44  4989.1 1801.87
  4995.0 1796.90  4995.5 1796.40  5005.1 1796.90  5011.1 1800.85  5080.7 1801.75
  5789.1 1803.96  5953.1 1804.20  5974.7 1811.94  5984.8 1811.92  6019.5 1798.83
  6043.3 1796.90  6104.7 1805.51  6225.4 1805.31  6371.8 1806.35  6732.7 1815.01
#Mann=15,-1,0
  2181.9   0.035       0  2279.9   0.094       0  2397.4   0.035       0
  2440.4   0.045       0  2677.3    0.07       0  2976.7   0.045       0
  3508.8    0.07       0  3836.3   0.035       0  4030.7    0.07       0
  4995.0    0.07       0  5005.1    0.07       0  5080.7   0.045       0
  5789.1    0.07       0  6225.4   0.045       0  6371.8    0.07       0
Bank Sta=4995,5005.1
Exp/Cntr=0.3,0.1

Type RM Length L Ch R = 1,18611,1463,1463,1463
BEGIN DESCRIPTION:
Tributary No. 1 to Elm Creek 21.0
END DESCRIPTION:
XS GIS Cut Line= 3
      1560255.00      6827888.00      1562361.72      6825801.39
      1562882.21      6824659.04
#Sta/Elev= 30
  2172.8 1809.81  2949.4 1805.40  3642.5 1801.14  4258.8 1799.61  4620.6 1800.18
  4647.7 1801.19  4690.1 1798.02  4725.5 1800.37  4767.9 1800.35  4789.1 1798.31
  4824.5 1800.50  4930.6 1801.42  4973.0 1801.13  4994.2 1799.42  4994.9 1798.02
  4995.4 1797.52  5005.1 1798.02  5008.3 1800.86  5029.6 1800.16  5059.3 1801.61
  5278.8 1800.97  5482.3 1802.73  5702.1 1802.50  5911.0 1805.02  5934.1 1807.41
  5951.6 1806.46  5997.7 1807.04  6130.0 1810.68  6229.6 1813.17  6393.3 1814.28
#Mann=8,-1,0
  2172.8   0.045       0  2949.4    0.07       0  3642.5   0.045       0
  4620.6    0.07       0  4994.9    0.07       0  5005.1    0.07       0
  5059.3   0.045       0  6130.0   0.035       0
Bank Sta=4994.9,5005.1
Exp/Cntr=0.3,0.1

Type RM Length L Ch R = 1,17148,978,978,978
BEGIN DESCRIPTION:
Tributary No. 1 to Elm Creek 20.0
END DESCRIPTION:
XS GIS Cut Line= 3
      1560805.02      6828537.98      1562725.10      6826662.56
      1563615.64      6825571.98
#Sta/Elev= 30
  2453.4 1814.42  2467.9 1814.53  2580.6 1810.64  2659.6 1810.46  3089.5 1805.59
  3430.9 1801.73  3448.8 1801.36  3740.3 1798.82  4257.8 1797.50  4376.9 1798.78
  4504.2 1797.01  4652.6 1797.38  4702.2 1794.56  4751.6 1797.08  4797.7 1796.89
  4914.2 1797.02  4939.4 1795.72  4984.9 1795.69  4994.9 1794.33  4995.4 1793.83
  5005.1 1794.33  5013.2 1796.04  5020.4 1794.33  5034.5 1796.51  5062.8 1797.24
  5147.5 1796.11  5359.9 1797.34  5458.7 1798.31  5877.8 1802.47  6545.4 1811.23
#Mann=14,-1,0
  2453.4   0.063       0  2467.9   0.035       0  2659.6   0.045       0
  3089.5    0.07       0  3430.9   0.035       0  3448.8   0.045       0
  4257.8    0.07       0  4797.7    0.16       0  4939.4    0.07       0
  4994.9    0.07       0  5005.1    0.07       0  5359.9   0.035       0
  5458.7    0.07       0  5877.8   0.045       0
Bank Sta=4994.9,5005.1
Exp/Cntr=0.3,0.1

Type RM Length L Ch R = 1,16170,914,914,914
BEGIN DESCRIPTION:
Tributary No. 1 to Elm Creek 19.0
END DESCRIPTION:
XS GIS Cut Line= 3
      1562006.03      6828368.39      1563400.28      6827083.51
      1563850.68      6826503.96
#Sta/Elev= 30
  3245.3 1799.18  3436.8 1798.34  3972.4 1794.46  4062.2 1794.35  4093.2 1794.12
  4200.4 1792.91  4339.2 1794.29  4558.6 1793.87  4677.8 1793.81  4724.1 1792.14
  4745.1 1794.14  4830.2 1793.01  4992.9 1794.89  4994.4 1792.14  4994.9 1791.64
  5005.6 1792.14  5007.1 1794.88  5042.3 1792.46  5049.6 1794.60  5063.8 1795.30
  5098.7 1795.22  5141.1 1795.88  5162.2 1799.44  5191.2 1801.26  5198.9 1800.64
  5205.7 1797.02  5220.1 1795.78  5284.4 1795.70  5842.7 1806.49  5875.3 1806.87
#Mann=13,-1,0
  3245.3   0.045       0  3436.8    0.07       0  3972.4   0.035       0
  4062.2    0.07       0  4093.2   0.035       0  4200.4    0.07       0
  4339.2    0.16       0  4558.6    0.07       0  4677.8    0.16       0
  4994.4    0.07       0  5005.6    0.16       0  5098.7    0.07       0
  5842.7   0.035       0
Bank Sta=4994.4,5005.6
Exp/Cntr=0.3,0.1

Type RM Length L Ch R = 1,15256,989,989,989
BEGIN DESCRIPTION:
Tributary No. 1 to Elm Creek 18.0
END DESCRIPTION:
XS GIS Cut Line= 3
      1562608.01      6828691.52      1563747.14      6827731.20
      1564170.06      6827087.87
#Sta/Elev= 30
  3510.1 1799.32  3535.6 1798.91  3586.6 1797.76  3631.2 1797.45  3659.8 1795.67
  3849.3 1794.00  4319.1 1791.39  4382.8 1790.10  4454.3 1792.03  4482.9 1790.98
  4689.1 1790.77  4731.3 1790.00  4752.1 1791.03  4841.6 1791.02  4986.2 1790.44
  4993.9 1789.76  4994.2 1788.49  4994.7 1787.99  5005.8 1788.49  5007.5 1790.07
  5015.8 1789.94  5022.6 1788.49  5043.7 1791.76  5205.3 1792.58  5405.2 1794.22
  5605.6 1797.98  5658.3 1798.34  5709.5 1799.98  5721.9 1801.66  5769.9 1802.19
#Mann=10,-1,0
  3510.1   0.125       0  3535.6    0.07       0  3586.6   0.035       0
  3849.3    0.07       0  4689.1    0.16       0  4841.6    0.07       0
  4994.2    0.07       0  5005.8    0.07       0  5205.3   0.045       0
  5605.6   0.035       0
Bank Sta=4994.2,5005.8
Exp/Cntr=0.3,0.1

Type RM Length L Ch R = 1,14267,938,938,938
BEGIN DESCRIPTION:
Tributary No. 1 to Elm Creek 17.0
END DESCRIPTION:
XS GIS Cut Line= 3
      1562882.89      6829529.59      1563852.14      6828582.14
      1564559.50      6827566.01
#Sta/Elev= 30
  3644.6 1799.81  3661.4 1800.78  3675.5 1799.39  3880.6 1797.80  3915.9 1796.06
  4036.2 1794.39  4064.5 1794.98  4163.5 1792.52  4255.4 1792.22  4269.5 1792.97
  4425.1 1790.79  4849.5 1789.65  4913.0 1788.21  4948.3 1789.55  4969.6 1789.01
  4983.7 1786.35  4990.7 1787.60  4994.0 1786.35  4994.5 1785.85  5006.0 1786.35
  5012.5 1788.10  5134.6 1788.69  5155.6 1789.85  5191.3 1788.70  5343.2 1789.98
  5516.0 1789.93  5726.9 1792.72  5975.1 1797.60  6182.2 1799.17  6238.1 1799.77
#Mann=5,-1,0
  3644.6    0.07       0  4994.0    0.07       0  5006.0    0.07       0
  5726.9   0.045       0  6182.2    0.07       0
Bank Sta=4994,5006
Exp/Cntr=0.3,0.1

Type RM Length L Ch R = 1,13329,466,466,466
BEGIN DESCRIPTION:
Tributary No. 1 to Elm Creek 16.0
END DESCRIPTION:
XS GIS Cut Line= 3
      1563104.98      6829838.02      1564395.24      6828528.97
      1564759.65      6827762.19
#Sta/Elev= 30
  3048.6 1802.02  3212.5 1799.50  3303.1 1798.74  3494.1 1794.22  3727.4 1791.25
  3769.9 1791.61  3840.6 1789.95  4392.2 1787.91  4667.9 1788.00  4781.1 1786.67
  4788.2 1785.43  4795.2 1786.55  4802.3 1785.03  4809.4 1787.27  4816.5 1785.35
  4823.5 1787.19  4830.6 1787.54  4963.6 1786.35  4991.9 1787.09  4994.0 1785.03
  4994.5 1784.53  5006.1 1785.03  5014.6 1785.82  5020.6 1788.62  5031.6 1790.90
  5043.4 1790.70  5292.8 1793.01  5429.1 1792.83  5639.1 1797.62  5735.6 1798.54
#Mann=5,-1,0
  3048.6   0.035       0  3212.5    0.07       0  4994.0    0.07       0
  5006.1    0.07       0  5043.4   0.045       0
Bank Sta=4994,5006.1
Exp/Cntr=0.3,0.1

Type RM Length L Ch R = 1,12863,516,516,516
BEGIN DESCRIPTION:
Tributary No. 1 to Elm Creek 15.0
END DESCRIPTION:
XS GIS Cut Line= 3
      1563155.01      6830037.99      1564741.27      6828775.09
      1565255.00      6828088.00
#Sta/Elev= 30
  2972.4 1804.12  3000.4 1803.42  3036.3 1804.68  3079.9 1803.01  3086.6 1803.17
  3178.2 1799.87  3598.7 1794.85  3841.3 1789.84  4238.5 1787.29  4517.2 1787.28
  4558.8 1788.32  4630.9 1786.43  4651.7 1787.56  4972.0 1787.01  4992.8 1785.11
  4994.0 1783.40  4994.5 1782.90  5006.1 1783.40  5014.8 1785.61  5040.9 1786.08
  5082.1 1786.64  5151.5 1786.64  5185.7 1785.54  5200.3 1787.09  5328.9 1788.56
  5394.2 1788.76  5479.6 1791.51  5579.7 1792.19  5698.0 1795.23  5857.9 1797.97
#Mann=10,-1,0
  2972.4   0.063       0  3079.9   0.035       0  3086.6    0.07       0
  4994.0    0.07       0  5006.1    0.07       0  5040.9    0.16       0
  5082.1    0.07       0  5151.5    0.16       0  5328.9    0.07       0
  5698.0   0.045       0
Bank Sta=4994,5006.1
Exp/Cntr=0.3,0.1

Type RM Length L Ch R = 1,12347,436,436,436
BEGIN DESCRIPTION:
Tributary No. 1 to Elm Creek 14.0
END DESCRIPTION:
XS GIS Cut Line= 3
      1564299.30      6830026.14      1564939.41      6829405.22
      1565355.00      6828088.01
#Sta/Elev= 30
  3409.4 1789.64  3475.7 1789.26  3511.2 1788.18  3638.5 1786.92  4211.3 1784.84
  4400.4 1785.13  4654.8 1784.22  4696.7 1785.44  4831.4 1785.52  4854.0 1785.04
  4958.2 1785.52  4979.9 1785.13  4994.0 1783.29  4994.5 1782.79  5005.6 1782.79
  5006.1 1783.29  5021.8 1785.26  5042.8 1785.04  5074.2 1786.96  5109.9 1787.71
  5133.0 1788.97  5170.6 1789.39  5189.6 1790.58  5219.1 1790.48  5267.6 1791.47
  5332.3 1793.80  5344.2 1793.65  5524.4 1796.87  5605.8 1798.10  5682.4 1798.81
#Mann=9,-1,0
  3409.4    0.07       0  4958.2    0.16       0  4994.0    0.07       0
  5006.1    0.16       0  5109.9    0.07       0  5219.1   0.045       0
  5344.2    0.07       0  5524.4   0.045       0  5605.8    0.07       0
Bank Sta=4994,5006.1
Exp/Cntr=0.3,0.1

Type RM Length L Ch R = 1,11911,768,768,768
BEGIN DESCRIPTION:
Tributary No. 1 to Elm Creek 13.0
END DESCRIPTION:
XS GIS Cut Line= 4
      1564587.67      6829825.15      1565377.86      6829009.97
      1565475.70      6828941.45      1565712.06      6828455.43
#Sta/Elev= 30
  3832.2 1786.38  4479.0 1784.81  4662.9 1783.10  4733.5 1784.43  4747.5 1781.94
  4761.7 1781.25  4832.4 1783.03  4860.7 1781.24  4889.0 1784.05  4981.0 1784.77
  4988.4 1784.67  4993.9 1781.24  4994.4 1780.74  5006.1 1781.24  5010.6 1784.96
  5091.7 1784.45  5096.6 1785.78  5102.1 1784.69  5119.1 1787.39  5157.5 1787.87
  5192.3 1786.21  5260.0 1789.25  5299.5 1788.79  5327.7 1790.52  5344.6 1790.39
  5350.2 1792.51  5367.2 1792.00  5372.8 1793.21  5474.3 1795.09  5627.4 1797.35
#Mann=4,-1,0
  3832.2    0.07       0  4993.9    0.07       0  5006.1    0.07       0
  5474.3   0.045       0
Bank Sta=4993.9,5006.1
Exp/Cntr=0.3,0.1

Type RM Length L Ch R = 1,11143,787,787,787
BEGIN DESCRIPTION:
Tributary No. 1 to Elm Creek 12.0
END DESCRIPTION:
XS GIS Cut Line= 3
      1564486.64      6830558.81      1565608.07      6829308.60
      1565977.72      6828556.05
#Sta/Elev= 30
  3804.3 1790.68  3952.8 1789.78  4044.7 1787.85  4320.5 1786.59  4356.2 1785.62
  4483.5 1784.74  4773.6 1784.17  4893.9 1782.73  4972.4 1782.86  4979.1 1783.50
  4993.3 1782.24  4993.8 1779.41  4994.3 1778.91  5006.2 1779.41  5021.8 1781.72
  5135.3 1781.63  5184.7 1782.56  5262.5 1781.60  5407.5 1782.03  5707.3 1783.74
  5762.4 1785.43  5780.0 1786.13  5803.8 1787.45  5854.4 1787.68  5930.1 1789.76
  6116.4 1792.69  6185.8 1793.43  6259.2 1794.74  6313.3 1795.46  6322.2 1795.63
#Mann=10,-1,0
  3804.3    0.07       0  4993.8    0.07       0  5006.2    0.07       0
  5407.5   0.045       0  5762.4    0.07       0  5780.0   0.045       0
  6116.4    0.07       0  6185.8   0.045       0  6259.2    0.07       0
  6313.3   0.045       0
Bank Sta=4993.8,5006.2
Exp/Cntr=0.3,0.1

Type RM Length L Ch R = 1,10356,804,804,804
BEGIN DESCRIPTION:
Tributary No. 1 to Elm Creek 11.0
END DESCRIPTION:
XS GIS Cut Line= 3
      1565012.43      6831024.96      1565977.66      6829615.67
      1566290.47      6828584.94
#Sta/Elev= 30
  3324.4 1788.72  3640.3 1785.95  3676.2 1786.30  3849.5 1784.26  3986.9 1784.06
  4302.5 1781.72  4536.2 1781.63  4556.4 1781.53  4979.4 1780.41  4993.4 1780.05
  4993.8 1778.83  4994.3 1778.33  5006.3 1778.83  5006.4 1779.42  5015.3 1778.83
  5021.3 1780.59  5155.5 1781.75  5180.0 1783.05  5212.9 1782.68  5270.5 1784.10
  5311.6 1784.09  5406.3 1785.62  5427.2 1786.66  5458.8 1786.05  5544.8 1786.81
  5636.2 1788.54  5709.4 1788.46  5831.1 1790.41  5887.0 1790.39  6109.7 1792.94
#Mann=6,-1,0
  3324.4    0.07       0  4536.2   0.045       0  4556.4    0.07       0
  4993.8   0.045       0  5006.3    0.07       0  5544.8    0.07       0
Bank Sta=4993.8,5006.3
Exp/Cntr=0.3,0.1

Type RM Length L Ch R = 1,9552,1411,1411,1411
BEGIN DESCRIPTION:
Tributary No. 1 to Elm Creek 10.0
END DESCRIPTION:
XS GIS Cut Line= 3
      1565447.22      6831223.21      1566398.96      6830129.81
      1566848.08      6828695.27
#Sta/Elev= 30
  3550.4 1786.48  3673.2 1786.25  3708.4 1784.50  3878.2 1783.57  4168.8 1781.51
  4619.5 1780.59  4949.3 1779.55  4991.1 1778.90  4993.8 1776.67  4994.3 1776.17
  5006.3 1776.67  5054.3 1778.95  5172.8 1779.65  5180.0 1777.92  5205.3 1777.05
  5237.7 1779.92  5273.6 1779.65  5376.3 1779.41  5387.4 1779.49  5586.5 1780.54
  5630.6 1781.77  5670.1 1780.86  5759.0 1781.80  5892.6 1781.34  6145.4 1785.20
  6172.6 1786.96  6217.4 1784.17  6248.9 1787.01  6353.6 1787.30  6503.2 1789.83
#Mann=10,-1,0
  3550.4    0.07       0  3878.2   0.045       0  4619.5    0.07       0
  4993.8    0.07       0  5006.3    0.07       0  5273.6   0.045       0
  5376.3   0.035       0  5387.4    0.07       0  5586.5   0.045       0
  5759.0    0.07       0
Bank Sta=4993.8,5006.3
Exp/Cntr=0.3,0.1

Type RM Length L Ch R = 1,8141,481,481,481
BEGIN DESCRIPTION:
Tributary No. 1 to Elm Creek 9.0
END DESCRIPTION:
XS GIS Cut Line= 3
      1565934.78      6831303.73      1567249.32      6830140.66
      1567670.17      6829107.49
#Sta/Elev= 30
  3244.8 1784.82  3673.7 1780.80  4261.8 1779.40  4481.8 1778.18  4567.0 1776.94
  4623.1 1777.97  4685.8 1777.43  4736.9 1777.88  4906.7 1776.90  4956.0 1776.32
  4963.6 1775.82  4970.2 1774.32  4992.0 1774.64  4993.6 1773.91  4994.1 1773.41
  5006.4 1773.91  5013.7 1777.02  5067.7 1780.09  5154.0 1780.26  5212.3 1781.47
  5337.6 1783.42  5423.1 1782.98  5437.2 1783.21  5553.3 1784.18  5558.7 1785.12
  5588.2 1786.05  5726.3 1785.39  5866.7 1786.71  6028.7 1789.65  6115.6 1790.03
#Mann=7,-1,0
  3244.8   0.045       0  4685.8    0.07       0  4993.6    0.07       0
  5006.4    0.07       0  5212.3   0.045       0  5423.1    0.07       0
  5437.2   0.045       0
Bank Sta=4993.6,5006.4
Exp/Cntr=0.3,0.1

Type RM Length L Ch R = 1,7660,721,721,721
BEGIN DESCRIPTION:
Tributary No. 1 to Elm Creek 8.0
END DESCRIPTION:
XS GIS Cut Line= 3
      1566310.99      6831288.25      1567494.19      6830528.37
      1567983.14      6829904.04
#Sta/Elev= 30
  3593.8 1783.72  3800.6 1780.46  3864.3 1780.64  4015.6 1779.28  4145.7 1779.48
  4218.4 1778.15  4327.4 1778.13  4406.7 1777.11  4733.0 1777.00  4769.3 1776.04
  4811.3 1776.04  4941.7 1776.72  4950.9 1775.89  4972.1 1775.75  4978.0 1775.26
  4987.3 1773.12  4993.6 1773.04  4994.1 1772.54  5006.0 1772.54  5006.5 1773.04
  5008.1 1775.82  5014.5 1776.34  5043.4 1777.24  5105.8 1776.98  5138.1 1777.27
  5261.4 1778.48  5483.2 1780.27  5535.0 1780.57  5609.0 1781.50  5793.0 1782.54
#Mann=10,-1,0
  3593.8   0.045       0  4811.3    0.07       0  4993.6    0.07       0
  5006.5    0.07       0  5105.8   0.045       0  5138.1    0.07       0
  5261.4   0.045       0  5483.2    0.07       0  5535.0   0.045       0
  5609.0    0.07       0
Bank Sta=4993.6,5006.5
Exp/Cntr=0.3,0.1

Type RM Length L Ch R = 1,6939,337,337,337
BEGIN DESCRIPTION:
Tributary No. 1 to Elm Creek 7.0
END DESCRIPTION:
XS GIS Cut Line= 3
      1566704.95      6831965.13      1567712.09      6831000.35
      1568384.96      6830402.47
#Sta/Elev= 30
  3849.6 1786.63  3909.2 1786.70  3913.6 1786.71  4050.0 1786.88  4051.2 1786.85
  4137.7 1786.38  4253.1 1784.31  4298.7 1783.33  4430.8 1780.00  4601.8 1778.86
  4682.1 1776.47  4717.6 1777.14  4739.5 1776.67  4754.3 1776.56  4877.1 1775.65
  4888.3 1775.60  4915.7 1775.74  4951.0 1773.73  4957.9 1774.37  4979.3 1773.09
  4986.2 1773.89  4993.5 1773.09  4994.0 1772.59  5006.6 1773.09  5007.6 1774.96
  5035.9 1776.44  5134.9 1774.94  5222.8 1775.02  5751.0 1776.25  6144.4 1779.01
#Mann=16,-1,0
  3849.6   0.045       0  3909.2   0.035       0  3913.6   0.045       0
  4050.0   0.035       0  4051.2   0.045       0  4253.1   0.035       0
  4298.7   0.045       0  4430.8   0.035       0  4601.8    0.07       0
  4739.5   0.045       0  4754.3    0.07       0  4877.1   0.045       0
  4888.3    0.07       0  4993.5    0.07       0  5006.6    0.07       0
  5222.8   0.045       0
Bank Sta=4993.5,5006.6
Exp/Cntr=0.3,0.1

Type RM Length L Ch R = 1,6602,934,934,934
BEGIN DESCRIPTION:
Tributary No. 1 to Elm Creek 6.0
END DESCRIPTION:
XS GIS Cut Line= 3
      1567074.85      6832176.92      1567853.52      6831301.60
      1568916.40      6830390.32
#Sta/Elev= 30
  3994.2 1784.31  4086.0 1783.33  4170.4 1780.18  4223.3 1780.23  4369.3 1778.85
  4623.7 1779.06  4637.9 1778.23  4657.3 1774.05  4829.2 1773.80  4857.8 1777.26
  4878.7 1774.82  4935.6 1774.18  4960.6 1772.29  4993.5 1772.17  4994.0 1771.67
  5006.6 1772.17  5035.1 1775.14  5084.4 1776.15  5141.3 1774.83  5365.5 1774.66
  5434.0 1774.65  5511.3 1775.16  5567.6 1774.89  5657.2 1774.97  5701.2 1774.84
  5803.0 1775.72  5842.8 1778.18  5871.4 1778.35  5948.8 1775.60  6565.8 1777.10
#Mann=16,-1,0
  3994.2   0.035       0  4223.3   0.063       0  4369.3   0.035       0
  4657.3    0.07       0  4829.2   0.035       0  4960.6    0.07       0
  4993.5    0.07       0  5006.6    0.07       0  5365.5   0.035       0
  5434.0    0.07       0  5511.3   0.035       0  5567.6    0.07       0
  5657.2   0.035       0  5701.2    0.07       0  5803.0   0.063       0
  5948.8   0.035       0
Bank Sta=4993.5,5006.6
Exp/Cntr=0.3,0.1

Type RM Length L Ch R = 1,5668,772,772,772
BEGIN DESCRIPTION:
Tributary No. 1 to Elm Creek 5.6
END DESCRIPTION:
XS GIS Cut Line= 3
      1567729.85      6832613.41      1568907.83      6831463.84
      1569297.54      6830952.96
#Sta/Elev= 30
  3960.0 1780.52  3987.4 1780.72  4002.8 1779.32  4024.0 1779.32  4031.1 1778.01
  4058.9 1778.21  4137.1 1777.10  4151.3 1778.40  4172.6 1776.57  4207.2 1776.57
  4264.4 1773.84  4413.1 1772.50  4547.3 1774.20  4717.1 1772.48  4830.3 1774.46
  4929.3 1773.14  4939.2 1771.96  4971.7 1772.14  4993.4 1770.35  4993.9 1769.85
  5006.6 1770.35  5042.4 1772.16  5113.0 1773.09  5433.2 1772.11  5537.3 1772.12
  5638.9 1773.86  5664.4 1773.34  5714.3 1774.97  5871.7 1774.22  6248.5 1775.88
#Mann=10,-1,0
  3960.0   0.094       0  3987.4   0.125       0  4058.9   0.094       0
  4207.2   0.063       0  4939.2    0.07       0  4993.4    0.07       0
  5006.6    0.07       0  5433.2   0.035       0  5638.9    0.07       0
  5871.7   0.045       0
Bank Sta=4993.4,5006.6
Exp/Cntr=0.3,0.1

Type RM Length L Ch R = 1,4896,563,563,563
BEGIN DESCRIPTION:
Tributary No. 1 to Elm Creek 5.3
END DESCRIPTION:
XS GIS Cut Line= 3
      1567910.42      6833058.29      1569192.16      6832212.10
      1569751.52      6831600.88
#Sta/Elev= 30
  3547.2 1773.73  3587.9 1772.47  3593.9 1773.14  3624.0 1772.06  3660.2 1771.81
  3831.7 1772.47  3901.9 1771.59  3925.0 1772.09  3955.1 1771.15  4053.1 1771.30
  4105.6 1771.93  4114.7 1771.30  4179.3 1771.19  4755.8 1771.67  4879.3 1770.92
  4942.7 1771.12  4966.6 1770.92  4993.4 1769.84  4993.9 1769.34  5006.2 1769.34
  5006.7 1769.84  5050.8 1770.96  5186.9 1770.60  5371.3 1771.63  5378.1 1771.09
  5413.9 1772.04  5434.8 1771.70  5470.0 1772.62  5501.5 1772.60  5911.6 1775.15
#Mann=8,-1,0
  3547.2   0.094       0  3660.2   0.063       0  3901.9   0.094       0
  4053.1   0.063       0  4179.3    0.07       0  4993.4    0.07       0
  5006.7    0.07       0  5501.5   0.045       0
Bank Sta=4993.4,5006.7
Exp/Cntr=0.3,0.1

Type RM Length L Ch R = 1,4333,983,983,983
BEGIN DESCRIPTION:
Tributary No. 1 to Elm Creek 5.0
END DESCRIPTION:
XS GIS Cut Line= 4
      1567871.70      6833335.03      1568442.20      6832981.20
      1569404.29      6832705.96      1570055.64      6832599.46
#Sta/Elev= 30
  3328.0 1776.07  3334.8 1774.91  3351.1 1774.95  3414.3 1775.01  3444.7 1772.88
  3475.9 1772.41  3529.1 1771.90  3594.5 1772.50  3649.1 1773.09  3697.4 1772.75
  3707.1 1773.26  3749.4 1772.43  3755.5 1773.14  3837.9 1772.96  3895.9 1770.86
  3917.2 1771.42  3950.1 1770.67  4180.3 1770.36  4907.1 1770.42  4993.3 1768.68
  4993.8 1768.18  5006.2 1768.18  5006.7 1768.68  5041.3 1769.96  5093.9 1770.31
  5355.4 1770.20  5568.2 1770.95  5598.6 1773.71  5614.8 1774.19  5660.0 1773.31
#Mann=12,-1,0
  3328.0   0.045       0  3351.1   0.094       0  3475.9    0.07       0
  3529.1   0.063       0  3594.5   0.035       0  3707.1   0.063       0
  3950.1   0.035       0  4180.3    0.07       0  4993.3    0.07       0
  5006.7    0.07       0  5093.9   0.045       0  5614.8    0.07       0
Bank Sta=4993.3,5006.7
Exp/Cntr=0.3,0.1

Type RM Length L Ch R = 1,3350,1046,1046,1046
BEGIN DESCRIPTION:
Tributary No. 1 to Elm Creek 4.5
END DESCRIPTION:
XS GIS Cut Line= 3
      1568138.94      6834013.61      1569429.44      6833193.63
      1570190.02      6832724.69
#Sta/Elev= 30
  3812.5 1771.63  4147.4 1769.70  4589.8 1769.82  4605.2 1767.87  4625.3 1766.99
  4807.0 1766.85  4839.7 1766.61  4929.9 1766.66  4959.3 1767.72  4972.3 1769.14
  4980.8 1767.87  4987.5 1769.44  4993.2 1766.51  4993.7 1766.01  5006.9 1766.51
  5016.3 1768.11  5024.0 1767.24  5029.9 1768.67  5045.1 1769.44  5118.0 1769.72
  5133.2 1770.30  5139.1 1771.73  5154.4 1771.21  5160.3 1772.54  5210.8 1769.83
  5233.1 1769.04  6147.8 1770.73  6178.6 1770.98  6217.2 1773.57  6235.0 1773.17
#Mann=9,-1,0
  3812.5   0.045       0  4605.2    0.07       0  4807.0   0.045       0
  4839.7    0.07       0  4959.3   0.035       0  4993.2   0.035       0
  5006.9   0.035       0  5210.8   0.045       0  6217.2    0.07       0
Bank Sta=4993.2,5006.9
Exp/Cntr=0.3,0.1

Type RM Length L Ch R = 1,2304,837,837,837
BEGIN DESCRIPTION:
Tributary No. 1 to Elm Creek 4.0
END DESCRIPTION:
XS GIS Cut Line= 3
      1569118.84      6834243.29      1569982.46      6833761.70
      1570256.38      6833578.24
#Sta/Elev= 30
  4087.5 1772.07  4337.6 1771.43  4593.2 1767.16  4624.4 1768.63  4765.0 1766.76
  4793.8 1767.15  4815.9 1767.21  4846.1 1765.32  4851.9 1766.87  4861.7 1766.70
  4867.9 1765.32  4873.6 1768.98  4883.9 1768.39  4889.6 1770.89  4896.0 1771.57
  4949.0 1772.26  4976.4 1769.44  4992.4 1762.67  4992.9 1758.65  4993.4 1758.15
  5007.1 1758.65  5010.5 1758.82  5014.2 1758.65  5030.1 1767.83  5035.9 1769.77
  5094.7 1769.46  5124.7 1770.49  5259.9 1770.87  5332.1 1772.06  5406.0 1771.55
#Mann=6,-1,0
  4087.5   0.045       0  4593.2    0.16       0  4793.8    0.07       0
  4992.9    0.07       0  5007.1    0.07       0  5010.5    0.16       0
Bank Sta=4992.9,5007.1
Exp/Cntr=0.3,0.1

Type RM Length L Ch R = 1,1467,488,488,488
BEGIN DESCRIPTION:
Tributary No. 1 to Elm Creek 3.0
END DESCRIPTION:
XS GIS Cut Line= 3
      1569322.26      6834541.35      1569894.10      6834478.37
      1570326.66      6834142.09
#Sta/Elev= 30
  4424.7 1770.26  4707.8 1767.63  4749.4 1768.65  4774.8 1767.96  4779.8 1768.72
  4910.4 1765.64  4930.5 1760.70  4940.5 1759.82  4956.7 1759.79  4961.7 1761.35
  4970.7 1761.68  4980.8 1759.54  4990.8 1755.09  4992.9 1755.09  4993.4 1754.59
  5006.6 1754.59  5007.1 1755.09  5008.1 1760.68  5014.4 1761.13  5022.6 1764.32
  5028.9 1763.91  5037.1 1766.84  5051.5 1768.34  5103.9 1768.03  5165.6 1768.67
  5186.4 1767.91  5271.5 1767.88  5346.0 1768.78  5418.0 1768.73  5547.9 1769.75
#Mann=7,-1,0
  4424.7   0.045       0  4707.8    0.07       0  4992.9    0.07       0
  5007.1    0.07       0  5103.9   0.035       0  5346.0    0.16       0
  5418.0    0.07       0
Bank Sta=4992.9,5007.1
Exp/Cntr=0.3,0.1

Type RM Length L Ch R = 1,979,459,459,459
BEGIN DESCRIPTION:
Tributary No. 1 to Elm Creek 2.0
END DESCRIPTION:
XS GIS Cut Line= 3
      1569938.94      6834997.76      1570223.79      6834757.27
      1570523.20      6834256.44
#Sta/Elev= 30
  4627.2 1770.30  4687.4 1769.45  4709.6 1769.78  4743.6 1768.26  4857.9 1766.71
  4865.6 1767.62  4900.8 1767.08  4950.2 1767.63  4972.2 1766.87  4978.8 1765.99
  4986.5 1762.86  4992.9 1754.82  4993.4 1754.32  5007.2 1754.82  5008.5 1764.53
  5014.4 1760.22  5022.4 1760.53  5035.8 1756.23  5045.5 1754.82  5051.3 1755.09
  5062.5 1758.85  5066.9 1760.59  5072.7 1764.98  5080.7 1766.21  5103.9 1767.22
  5131.1 1765.24  5146.6 1766.38  5189.4 1767.38  5358.7 1767.76  5583.5 1769.74
#Mann=6,-1,0
  4627.2    0.07       0  4687.4   0.035       0  4743.6    0.07       0
  4992.9    0.07       0  5007.2    0.07       0  5062.5   0.035       0
Bank Sta=4992.9,5007.2
Exp/Cntr=0.3,0.1
