--- Alkali Creek.prj (project) ---

Proj Title=Alkali Creek Base Level Engineering
Current Plan=p01
Default Exp/Contr=0.3,0.1
English Units
Geom File=g01
Flow File=f01
Plan File=p01
Y Axis Title=Elevation
X Axis Title(PF)=Main Channel Distance
X Axis Title(XS)=Station
BEGIN DESCRIPTION:
Alkali Creek
END DESCRIPTION:
DSS Export Rating Curves= 0
DSS Export Rating Curve Sorted= 0
DSS Export Volume Flow Curves= 0
DXF OffsetX= 0
DXF OffsetY= 0
DXF ScaleX= 1
DXF ScaleY= 10

--- Alkali Creek.p01 (plan) ---

Plan Title=Multiple Run
Short Identifier=Multiple
Geom File=g01
Flow File=f01
Subcritical Flow
K Sum by GR= 0
Std Step Tol= 0.01
Critical Tol= 0.01
Num of Std Step Trials= 20
Max Error Tol= 0.3
Flow Tol Ratio= 0.001
Split Flow NTrial= 30
Split Flow Tol= 0.02
Split Flow Ratio= 0.02
Log Output Level= 0
Friction Slope Method= 1
Unsteady Friction Slope Method= 2
Unsteady Bridges Friction Slope Method= 1
Parabolic Critical Depth
Global Vel Dist=  1 , 1 , 1
Global Log Level= 0
CheckData=True
Encroach Param= -1, 0, 0, 0
BEGIN DESCRIPTION:
Multiple Run
END DESCRIPTION:

--- Alkali Creek.f01 (steady flow) ---

Flow Title=Multiple
Program Version=4.10
Number of Profiles= 7
Profile Names=10-year,25-year,50-year,1pct_min,100-year,1pct_plu,500-year
River Rch & RM=Alkali Creek,Reach-1         ,100032
     304     437     550     344     687    1371    1088
River Rch & RM=Alkali Creek,Reach-1         ,97781
     815    1228    1596    1029    2054    4098    3449
River Rch & RM=Alkali Creek,Reach-1         ,92371
     843    1265    1640    1054    2102    4195    3505
River Rch & RM=Alkali Creek,Reach-1         ,85479
    1168    1772    2312    1494    2982    5949    5028
River Rch & RM=Alkali Creek,Reach-1         ,80246
    1186    1794    2335    1505    3004    5993    5039
River Rch & RM=Alkali Creek,Reach-1         ,72427
    1240    1876    2444    1576    3145    6275    5279
River Rch & RM=Alkali Creek,Reach-1         ,70826
    1240    1871    2433    1566    3124    6233    5222
River Rch & RM=Alkali Creek,Reach-1         ,66405
    1304    1970    2565    1652    3296    6577    5521
River Rch & RM=Alkali Creek,Reach-1         ,65314
    1344    2029    2641    1700    3391    6767    5673
River Rch & RM=Alkali Creek,Reach-1         ,60398
    1360    2052    2667    1715    3421    6826    5708
River Rch & RM=Alkali Creek,Reach-1         ,54921
    1395    2099    2724    1747    3486    6956    5793
River Rch & RM=Alkali Creek,Reach-1         ,51065
    1759    2668    3480    2243    4476    8930    7508
River Rch & RM=Alkali Creek,Reach-1         ,40455
    1849    2807    3665    2364    4717    9412    7924
River Rch & RM=Alkali Creek,Reach-1         ,38847
    1834    2779    3622    2333    4654    9287    7792
River Rch & RM=Alkali Creek,Reach-1         ,32414
    1938    2937    3830    2467    4922    9821    8243
River Rch & RM=Alkali Creek,Reach-1         ,26512
    1961    2971    3874    2495    4978    9932    8334
River Rch & RM=Alkali Creek,Reach-1         ,24367
    1970    2983    3889    2504    4996    9967    8358
River Rch & RM=Alkali Creek,Reach-1         ,22763
    2630    4015    5264    3407    6797   13562   11487
River Rch & RM=Alkali Creek,Reach-1         ,19387
    2621    3990    5218    3369    6721   13411   11302
Boundary for River Rch & Prof#=Alkali Creek,Reach-1         , 1
Up Type= 0
Dn Type= 3
Dn Slope=0.002
Boundary for River Rch & Prof#=Alkali Creek,Reach-1         , 2
Up Type= 0
Dn Type= 3
Dn Slope=0.002
Boundary for River Rch & Prof#=Alkali Creek,Reach-1         , 3
Up Type= 0
Dn Type= 3
Dn Slope=0.002
Boundary for River Rch & Prof#=Alkali Creek,Reach-1         , 4
Up Type= 0
Dn Type= 3
Dn Slope=0.002
Boundary for River Rch & Prof#=Alkali Creek,Reach-1         , 5
Up Type= 0
Dn Type= 3
Dn Slope=0.002
Boundary for River Rch & Prof#=Alkali Creek,Reach-1         , 6
Up Type= 0
Dn Type= 3
Dn Slope=0.002
Boundary for River Rch & Prof#=Alkali Creek,Reach-1         , 7
Up Type= 0
Dn Type= 3
Dn Slope=0.002
DSS Import GetInterval= 0
DSS Import GetPeak= 0
DSS Import FillOption= 0

--- Alkali Creek.g01 (geometry) ---

Geom Title=Existing Conditions

River Reach=Alkali Creek,Reach-1
Reach XY= 30
      1346705.00      6947638.00      1345905.00      6949038.00
      1347147.12      6949731.83      1348303.38      6952599.81
      1349205.50      6955858.24      1348457.01      6957232.17
      1349504.61      6957803.28      1348910.35      6958590.70
      1352511.51      6961136.37      1354664.83      6959998.52
      1354894.51      6963127.04      1355846.38      6962840.96
      1361321.03      6966037.84      1366208.39      6964795.76
      1368070.69      6966538.70      1370407.74      6966332.66
      1370809.63      6964942.63      1374344.31      6962988.74
      1375418.39      6965301.34      1376799.54      6965935.55
      1376515.76      6966947.68      1378014.80      6967098.48
      1378525.06      6968538.22      1383399.17      6965440.06
      1385906.45      6968334.47      1388181.94      6967514.14
      1388302.70      6970282.91      1391778.53      6970310.86
      1390855.98      6974177.74      1392555.00      6974488.00

Type RM Length L Ch R = 1,100032,434,434,434
BEGIN DESCRIPTION:
Alkali Creek 113.0
END DESCRIPTION:
XS GIS Cut Line= 3
      1346279.97      6947412.96      1346505.00      6947738.00
      1346686.53      6948173.01
#Sta/Elev= 30
  4600.6 2076.45  4651.3 2075.80  4866.2 2075.26  4937.8 2073.25  4946.6 2071.95
  4952.7 2071.90  4965.3 2069.63  4982.4 2064.90  4988.5 2063.81  4992.9 2062.21
  5005.1 2061.62  5008.6 2060.76  5008.8 2060.26  5012.3 2060.26  5012.6 2060.76
  5017.6 2062.37  5039.8 2064.47  5058.2 2067.93  5063.6 2067.58  5082.0 2069.83
  5087.4 2071.17  5100.0 2071.66  5135.1 2074.25  5158.5 2074.48  5234.3 2074.55
  5331.8 2073.79  5376.5 2074.26  5400.3 2073.65  5453.4 2074.54  5467.3 2073.88
#Mann=5,-1,0
  4600.6   0.035       0  4965.3    0.07       0  5008.6    0.07       0
  5012.6    0.07       0  5100.0   0.035       0
Bank Sta=5008.6,5012.6
Exp/Cntr=0.3,0.1

Type RM Length L Ch R = 1,99598,476,476,476
BEGIN DESCRIPTION:
Alkali Creek 112.0
END DESCRIPTION:
XS GIS Cut Line= 3
      1345929.97      6947762.99      1346155.00      6947888.00
      1346454.99      6948387.99
#Sta/Elev= 30
  4732.3 2074.13  4836.6 2072.72  4916.5 2073.17  4954.3 2071.69  4960.0 2068.59
  4976.0 2066.11  4981.7 2060.82  4986.9 2063.25  4992.6 2063.25  4997.5 2058.20
  5003.3 2062.46  5013.0 2059.87  5024.7 2059.99  5032.4 2055.82  5032.7 2055.32
  5036.4 2055.82  5040.3 2059.57  5048.0 2056.41  5055.8 2058.00  5071.4 2057.86
  5083.0 2062.01  5092.7 2069.56  5098.6 2069.05  5106.3 2071.96  5264.3 2072.55
  5456.2 2070.99  5506.7 2072.09  5522.3 2073.84  5528.1 2072.99  5572.8 2074.44
#Mann=5,-1,0
  4732.3   0.035       0  4836.6    0.07       0  5032.4    0.07       0
  5036.4    0.07       0  5264.3   0.035       0
Bank Sta=5032.4,5036.4
Exp/Cntr=0.3,0.1

Type RM Length L Ch R = 1,99122,422,422,422
BEGIN DESCRIPTION:
Alkali Creek 111.0
END DESCRIPTION:
XS GIS Cut Line= 3
      1345980.02      6948213.02      1346055.00      6948288.00
      1346400.04      6948481.21
#Sta/Elev= 30
  4894.2 2073.47  4929.5 2073.24  4972.0 2069.26  4986.1 2064.97  4996.7 2056.50
  5003.1 2056.50  5008.2 2054.20  5012.0 2053.74  5012.2 2053.24  5015.7 2053.24
  5016.0 2053.74  5023.2 2057.24  5045.9 2060.54  5051.6 2062.33  5067.6 2062.96
  5073.3 2065.44  5080.5 2065.11  5095.0 2066.85  5111.0 2067.75  5116.7 2068.61
  5126.3 2068.80  5138.4 2070.12  5169.8 2070.14  5206.5 2069.13  5213.7 2069.74
  5219.4 2069.03  5251.4 2068.73  5278.8 2071.71  5294.8 2072.63  5395.7 2072.41
#Mann=4,-1,0
  4894.2    0.07       0  5012.0    0.07       0  5016.0    0.07       0
  5169.8   0.035       0
Bank Sta=5012,5016
Exp/Cntr=0.3,0.1

Type RM Length L Ch R = 1,98700,414,414,414
BEGIN DESCRIPTION:
Alkali Creek 110.0
END DESCRIPTION:
XS GIS Cut Line= 3
      1345830.00      6948563.00      1346205.00      6948588.00
      1346530.00      6948613.00
#Sta/Elev= 30
  4628.3 2074.05  4643.3 2073.70  4663.4 2073.96  4693.4 2073.44  4703.5 2072.60
  4733.6 2072.27  4843.8 2069.40  4873.8 2067.68  4883.9 2066.74  4903.9 2062.28
  4924.0 2059.10  4934.0 2059.25  4954.0 2058.05  4984.1 2055.31  4994.1 2052.49
  4999.6 2049.92  4999.9 2049.42  5003.4 2049.42  5003.6 2049.92  5006.6 2049.92
  5034.2 2065.64  5044.3 2067.29  5054.3 2072.01  5064.3 2072.83  5077.6 2072.37
  5224.8 2072.41  5244.8 2073.15  5264.9 2074.64  5305.0 2074.61  5330.1 2075.16
#Mann=5,-1,0
  4628.3   0.035       0  4733.6    0.07       0  4999.6    0.07       0
  5003.6    0.07       0  5077.6   0.035       0
Bank Sta=4999.6,5003.6
Exp/Cntr=0.3,0.1

Type RM Length L Ch R = 1,98286,505,505,505
BEGIN DESCRIPTION:
Alkali Creek 109.0
END DESCRIPTION:
XS GIS Cut Line= 3
      1345830.00      6948663.00      1345974.86      6948867.62
      1346230.01      6948963.00
#Sta/Elev= 30
  4749.3 2071.63  4820.7 2070.37  4895.5 2067.24  4927.7 2065.54  4936.4 2063.88
  4942.5 2065.05  4951.2 2062.84  4957.3 2059.98  4963.7 2055.50  4972.1 2052.76
  4978.2 2052.48  4986.8 2049.32  4991.0 2049.05  4991.2 2048.55  4994.7 2048.55
  4995.0 2049.05  4997.2 2051.21  5010.4 2051.86  5015.8 2058.11  5021.5 2061.14
  5032.2 2063.02  5040.7 2065.39  5064.2 2066.51  5071.0 2067.71  5096.0 2068.15
  5101.3 2067.65  5181.5 2072.86  5186.8 2072.32  5230.0 2072.78  5272.4 2072.75
#Mann=5,-1,0
  4749.3   0.035       0  4895.5    0.07       0  4991.0    0.07       0
  4995.0    0.07       0  5230.0   0.035       0
Bank Sta=4991,4995
Exp/Cntr=0.3,0.1

Type RM Length L Ch R = 1,97781,495,495,495
BEGIN DESCRIPTION:
Alkali Creek 108.0
END DESCRIPTION:
XS GIS Cut Line= 3
      1345816.32      6949525.09      1346155.00      6949138.00
      1346480.03      6948812.97
#Sta/Elev= 30
  4489.8 2074.49  4494.0 2075.58  4543.8 2074.83  4550.9 2074.14  4653.8 2073.47
  4780.7 2072.75  4841.4 2069.94  4869.8 2065.60  4884.1 2064.34  4890.7 2064.83
  4907.7 2061.56  4911.6 2060.63  4919.2 2060.87  4925.8 2057.25  4933.4 2055.58
  4968.5 2050.96  4976.1 2047.79  4982.8 2048.78  4992.5 2045.91  4993.0 2045.41
  5001.6 2045.91  5004.1 2048.25  5007.7 2048.25  5018.3 2059.75  5032.4 2064.65
  5103.1 2070.86  5190.4 2072.86  5302.3 2073.04  5318.3 2073.07  5463.8 2073.31
#Mann=10,-1,0
  4489.8   0.045       0  4543.8   0.035       0  4653.8    0.07       0
  4780.7   0.035       0  4907.7    0.07       0  4992.5    0.07       0
  5001.6    0.07       0  5190.4   0.035       0  5302.3    0.07       0
  5318.3   0.035       0
Bank Sta=4992.5,5001.6
Exp/Cntr=0.3,0.1

Type RM Length L Ch R = 1,97286,467,467,467
BEGIN DESCRIPTION:
Alkali Creek 107.0
END DESCRIPTION:
XS GIS Cut Line= 3
      1346250.38      6949809.34      1346505.00      6949488.00
      1346955.67      6948958.65
#Sta/Elev= 30
  4585.9 2071.08  4623.9 2070.76  4716.9 2071.70  4765.6 2071.83  4839.1 2071.45
  4932.1 2070.37  4945.4 2068.66  4953.4 2065.37  4967.9 2052.47  4984.1 2044.53
  4984.6 2044.03  4993.2 2044.53  4995.9 2047.06  4999.2 2047.06  5003.0 2049.90
  5023.9 2049.94  5066.7 2054.75  5095.3 2061.19  5116.1 2059.82  5123.8 2061.73
  5144.7 2061.07  5194.1 2064.16  5211.5 2063.36  5258.6 2067.35  5337.1 2068.89
  5408.4 2069.03  5462.6 2069.55  5566.5 2070.99  5593.2 2071.24  5691.1 2072.00
#Mann=13,-1,0
  4585.9   0.045       0  4623.9   0.035       0  4716.9    0.07       0
  4765.6   0.045       0  4839.1    0.07       0  4984.1    0.07       0
  4993.2    0.07       0  5211.5   0.035       0  5337.1    0.07       0
  5408.4   0.035       0  5462.6    0.07       0  5566.5   0.035       0
  5593.2    0.07       0
Bank Sta=4984.1,4993.2
Exp/Cntr=0.3,0.1

Type RM Length L Ch R = 1,96819,463,463,463
BEGIN DESCRIPTION:
Alkali Creek 106.0
END DESCRIPTION:
XS GIS Cut Line= 3
      1346686.54      6949913.56      1346955.00      6949538.00
      1347148.77      6949299.42
#Sta/Elev= 30
  4538.3 2070.19  4724.0 2069.72  4805.8 2067.01  4841.4 2064.32  4900.4 2061.79
  4921.3 2060.21  4927.4 2058.82  4936.0 2059.30  4942.2 2054.45  4950.8 2056.91
  4956.9 2054.09  4963.1 2049.75  4974.7 2047.99  4986.4 2046.73  4992.3 2043.85
  4992.8 2043.35  5001.5 2043.85  5007.1 2045.06  5027.9 2045.97  5035.9 2047.28
  5056.7 2053.48  5091.9 2059.73  5120.6 2061.37  5128.5 2063.20  5135.0 2063.14
  5149.4 2066.20  5155.8 2065.42  5163.7 2066.79  5217.4 2069.26  5307.3 2071.72
#Mann=6,-1,0
  4538.3   0.045       0  4724.0   0.035       0  4974.7    0.07       0
  4992.3    0.07       0  5001.5    0.07       0  5217.4   0.035       0
Bank Sta=4992.3,5001.5
Exp/Cntr=0.3,0.1

Type RM Length L Ch R = 1,96356,432,432,432
BEGIN DESCRIPTION:
Alkali Creek 105.0
END DESCRIPTION:
XS GIS Cut Line= 3
      1346777.74      6950045.90      1347205.00      6949888.00
      1347521.01      6949694.99
#Sta/Elev= 30
  4548.6 2069.09  4606.4 2069.17  4639.9 2069.66  4731.1 2067.96  4817.1 2063.71
  4842.1 2061.24  4847.5 2061.70  4861.7 2059.53  4897.5 2056.18  4903.0 2053.76
  4908.3 2055.11  4918.8 2053.55  4940.1 2048.16  4950.8 2046.44  4972.1 2046.25
  4978.1 2040.77  4978.6 2040.27  4987.4 2040.77  4988.9 2042.36  4994.2 2042.90
  5001.4 2047.05  5007.0 2047.05  5017.7 2055.65  5027.3 2059.52  5069.9 2064.07
  5091.2 2065.00  5149.3 2070.10  5339.0 2075.34  5367.8 2074.50  5374.4 2074.09
#Mann=6,-1,0
  4548.6   0.045       0  4606.4   0.035       0  4861.7    0.07       0
  4978.1    0.07       0  4987.4    0.07       0  5367.8   0.035       0
Bank Sta=4978.1,4987.4
Exp/Cntr=0.3,0.1

Type RM Length L Ch R = 1,95924,448,448,448
BEGIN DESCRIPTION:
Alkali Creek 104.0
END DESCRIPTION:
XS GIS Cut Line= 3
      1347003.42      6950397.46      1347305.00      6950288.00
      1347595.86      6949959.09
#Sta/Elev= 30
  4674.2 2067.61  4909.9 2067.48  4923.8 2066.57  4931.2 2064.44  4963.1 2058.88
  4965.8 2057.58  4973.8 2053.71  4987.7 2039.93  4988.2 2039.43  4997.0 2039.93
  5023.0 2046.88  5044.8 2048.13  5065.7 2047.98  5094.1 2050.78  5101.7 2053.38
  5108.4 2051.71  5122.6 2056.03  5151.0 2059.91  5193.7 2062.19  5214.6 2062.28
  5235.5 2064.35  5278.2 2064.21  5320.8 2065.32  5342.1 2067.65  5363.5 2067.14
  5398.6 2067.74  5412.8 2068.50  5420.4 2069.76  5427.1 2069.17  5434.1 2070.37
#Mann=5,-1,0
  4674.2   0.035       0  4965.8    0.07       0  4987.7    0.07       0
  4997.0    0.07       0  5278.2   0.035       0
Bank Sta=4987.7,4997
Exp/Cntr=0.3,0.1

Type RM Length L Ch R = 1,95476,480,480,480
BEGIN DESCRIPTION:
Alkali Creek 103.0
END DESCRIPTION:
XS GIS Cut Line= 3
      1347066.33      6950512.49      1347655.00      6950538.00
      1348211.10      6950501.71
#Sta/Elev= 30
  4414.8 2066.79  4503.5 2066.34  4577.3 2063.31  4678.1 2060.02  4701.0 2059.33
  4783.8 2058.28  4888.7 2054.23  4944.0 2043.57  4984.0 2044.76  4994.0 2040.84
  5009.3 2038.24  5009.8 2037.74  5018.7 2038.24  5024.1 2050.25  5044.1 2061.24
  5080.0 2066.28  5124.3 2066.40  5184.4 2062.51  5204.4 2062.41  5224.5 2060.35
  5231.9 2057.29  5254.6 2052.79  5284.6 2051.80  5424.9 2054.59  5434.9 2055.14
  5465.0 2060.26  5505.1 2061.98  5535.1 2065.31  5553.2 2064.83  5561.3 2065.12
#Mann=7,-1,0
  4414.8   0.035       0  4577.3    0.07       0  4678.1   0.035       0
  4701.0    0.07       0  5009.3    0.07       0  5018.7    0.07       0
  5553.2   0.035       0
Bank Sta=5009.3,5018.7
Exp/Cntr=0.3,0.1

Type RM Length L Ch R = 1,94996,382,382,382
BEGIN DESCRIPTION:
Alkali Creek 102.0
END DESCRIPTION:
XS GIS Cut Line= 4
      1346742.74      6950743.34      1347355.00      6950838.00
      1347515.91      6950876.35      1348191.16      6950856.22
#Sta/Elev= 30
  4391.6 2067.04  4414.3 2066.97  4768.3 2065.53  4874.6 2058.51  4914.0 2055.41
  4930.2 2048.61  4972.3 2036.33  4972.8 2035.83  4981.9 2036.33  4982.1 2038.92
  4990.9 2041.53  5034.8 2042.38  5062.5 2044.88  5124.2 2056.45  5161.1 2059.76
  5166.3 2058.56  5284.9 2064.29  5325.7 2065.44  5415.7 2060.24  5465.8 2049.94
  5515.8 2043.00  5545.8 2046.51  5565.8 2052.20  5585.8 2050.09  5605.8 2052.56
  5615.8 2054.31  5622.7 2057.64  5627.7 2054.90  5705.9 2060.64  5852.1 2064.21
#Mann=5,-1,0
  4391.6   0.045       0  4414.3   0.035       0  4874.6    0.07       0
  4972.3    0.07       0  4981.9    0.07       0
Bank Sta=4972.3,4981.9
Exp/Cntr=0.3,0.1

Type RM Length L Ch R = 1,94614,503,503,503
BEGIN DESCRIPTION:
Alkali Creek 101.0
END DESCRIPTION:
XS GIS Cut Line= 3
      1346998.80      6951040.65      1347405.00      6951138.00
      1348194.57      6950995.07
#Sta/Elev= 30
  4631.8 2061.70  4743.8 2063.28  4905.5 2065.21  4957.0 2061.26  4967.2 2053.67
  4977.5 2043.28  4983.9 2040.74  4989.0 2044.11  5008.4 2038.24  5013.8 2034.21
  5014.3 2033.71  5023.4 2034.21  5025.9 2036.35  5039.2 2034.21  5059.7 2039.33
  5090.1 2041.86  5181.6 2044.05  5201.9 2049.46  5262.9 2056.25  5305.4 2058.00
  5358.9 2057.24  5417.4 2052.27  5465.8 2041.42  5496.7 2040.34  5517.0 2043.37
  5537.3 2050.56  5577.8 2058.91  5748.4 2065.00  5821.9 2063.52  5851.9 2065.92
#Mann=4,-1,0
  4631.8   0.045       0  4743.8    0.07       0  5013.8    0.07       0
  5023.4    0.07       0
Bank Sta=5013.8,5023.4
Exp/Cntr=0.3,0.1

Type RM Length L Ch R = 1,94111,434,434,434
BEGIN DESCRIPTION:
Alkali Creek 100.0
END DESCRIPTION:
XS GIS Cut Line= 3
      1347014.01      6951179.54      1347755.00      6951288.00
      1348207.54      6951329.28
#Sta/Elev= 30
  4255.4 2059.70  4334.8 2061.03  4377.7 2063.23  4415.2 2063.24  4420.3 2064.71
  4438.3 2063.50  4529.3 2064.94  4569.7 2064.10  4610.4 2060.34  4680.9 2056.28
  4694.8 2057.19  4719.7 2054.29  4741.5 2052.33  4759.6 2053.48  4822.4 2047.60
  4834.6 2048.27  4943.6 2040.15  5006.8 2039.48  5029.1 2034.35  5029.6 2033.85
  5039.8 2034.35  5044.5 2038.19  5054.4 2042.83  5059.4 2041.44  5064.5 2047.88
  5074.6 2052.58  5104.7 2057.87  5163.5 2060.58  5215.2 2062.06  5458.7 2062.94
#Mann=7,-1,0
  4255.4   0.045       0  4334.8    0.07       0  4610.4   0.035       0
  4719.7    0.07       0  5029.1    0.07       0  5039.8    0.07       0
  5163.5   0.035       0
Bank Sta=5029.1,5039.8
Exp/Cntr=0.3,0.1

Type RM Length L Ch R = 1,93677,448,448,448
BEGIN DESCRIPTION:
Alkali Creek 99.0
END DESCRIPTION:
XS GIS Cut Line= 3
      1346799.16      6951309.76      1347655.00      6951688.00
      1348426.76      6951860.97
#Sta/Elev= 30
  4064.3 2063.58  4275.8 2058.82  4364.8 2058.46  4468.9 2054.88  4617.1 2054.51
  4676.8 2054.35  4689.6 2056.46  4695.1 2054.19  4886.9 2050.95  4945.3 2045.26
  4962.3 2039.83  4978.1 2037.75  4985.6 2033.76  4985.7 2031.24  4986.2 2030.74
  4996.4 2031.24  4997.3 2033.49  5002.6 2033.49  5010.2 2037.05  5030.7 2037.88
  5051.2 2044.67  5100.8 2055.68  5133.2 2061.09  5251.3 2061.60  5317.7 2061.44
  5439.1 2057.02  5539.9 2057.99  5578.6 2058.82  5681.6 2061.11  5790.9 2062.25
#Mann=11,-1,0
  4064.3   0.045       0  4275.8    0.07       0  4617.1   0.035       0
  4676.8    0.07       0  4985.7    0.07       0  4996.4    0.07       0
  5100.8   0.035       0  5439.1    0.07       0  5539.9   0.035       0
  5578.6    0.07       0  5681.6   0.035       0
Bank Sta=4985.7,4996.4
Exp/Cntr=0.3,0.1

Type RM Length L Ch R = 1,93229,443,443,443
BEGIN DESCRIPTION:
Alkali Creek 98.0
END DESCRIPTION:
XS GIS Cut Line= 3
      1347070.36      6952323.22      1347505.00      6952088.00
      1347858.12      6951997.69
#Sta/Elev= 30
  4506.0 2066.64  4579.5 2064.54  4794.4 2061.98  4822.8 2060.59  4839.0 2061.14
  4844.7 2060.12  4875.1 2060.46  4897.9 2058.68  4904.6 2057.86  4910.3 2055.32
  4920.6 2055.71  4926.5 2049.74  4932.2 2046.05  4940.2 2044.68  4954.7 2042.74
  4970.2 2037.78  4986.4 2034.67  4991.8 2029.58  4992.3 2029.08  5002.9 2029.58
  5010.5 2034.26  5018.0 2036.08  5041.5 2037.16  5051.8 2040.48  5072.5 2043.39
  5113.8 2047.07  5204.1 2051.66  5217.0 2051.92  5303.8 2059.73  5364.7 2057.81
#Mann=6,-1,0
  4506.0    0.07       0  4794.4   0.035       0  4940.2    0.07       0
  4991.8    0.07       0  5002.9    0.07       0  5204.1   0.035       0
Bank Sta=4991.8,5002.9
Exp/Cntr=0.3,0.1

Type RM Length L Ch R = 1,92786,415,415,415
BEGIN DESCRIPTION:
Alkali Creek 97.0
END DESCRIPTION:
XS GIS Cut Line= 3
      1347361.24      6952644.35      1347805.00      6952338.00
      1348296.57      6952045.40
#Sta/Elev= 30
  4454.8 2062.46  4459.9 2062.48  4533.0 2059.45  4705.5 2058.86  4759.0 2058.91
  4836.1 2057.63  4872.5 2051.18  4879.1 2054.31  4900.1 2044.91  4909.8 2043.32
  4914.9 2040.11  4944.7 2035.63  4960.1 2029.31  4960.6 2028.81  4971.2 2029.31
  4971.7 2032.72  5017.3 2034.19  5029.1 2040.25  5060.3 2038.75  5066.1 2041.21
  5081.7 2039.99  5087.5 2042.87  5124.5 2044.63  5133.7 2041.96  5140.1 2036.98
  5149.0 2040.86  5177.1 2047.16  5235.5 2051.24  5455.9 2059.31  5566.1 2061.13
#Mann=9,-1,0
  4454.8   0.045       0  4459.9   0.035       0  4705.5    0.07       0
  4759.0   0.035       0  4909.8    0.07       0  4960.1    0.07       0
  4971.2    0.07       0  5149.0   0.035       0  5455.9    0.07       0
Bank Sta=4960.1,4971.2
Exp/Cntr=0.3,0.1

Type RM Length L Ch R = 1,92371,376,376,376
BEGIN DESCRIPTION:
Alkali Creek 96.0
END DESCRIPTION:
XS GIS Cut Line= 3
      1347645.50      6952787.60      1348155.00      6952538.00
      1348424.59      6952223.35
#Sta/Elev= 30
  4427.8 2057.44  4458.0 2058.17  4486.1 2057.25  4494.1 2058.13  4508.6 2057.01
  4615.5 2056.61  4683.0 2054.86  4694.5 2055.57  4705.5 2054.44  4711.1 2055.29
  4733.6 2052.87  4868.6 2046.96  4936.1 2042.78  4958.6 2037.91  4964.2 2033.90
  4995.2 2031.37  4996.6 2027.17  4997.1 2026.67  5007.9 2027.17  5016.6 2031.46
  5023.1 2031.95  5030.8 2034.25  5037.4 2033.97  5045.1 2037.40  5065.9 2041.06
  5080.2 2046.87  5094.5 2050.24  5101.1 2055.03  5193.3 2058.52  5409.5 2058.96
#Mann=3,-1,0
  4427.8    0.07       0  4996.6    0.07       0  5007.9    0.07       0
Bank Sta=4996.6,5007.9
Exp/Cntr=0.3,0.1

Type RM Length L Ch R = 1,91995,509,509,509
BEGIN DESCRIPTION:
Alkali Creek 95.0
END DESCRIPTION:
XS GIS Cut Line= 3
      1347502.22      6952863.57      1348288.65      6952805.11
      1348849.87      6952685.62
#Sta/Elev= 30
  4211.4 2057.83  4266.5 2057.43  4500.3 2056.22  4575.2 2056.00  4622.0 2054.68
  4627.0 2055.33  4645.4 2053.41  4795.8 2046.13  4892.3 2038.06  4926.2 2036.42
  4956.2 2031.50  4966.3 2031.94  4976.3 2029.28  4980.6 2026.79  4981.1 2026.29
  4992.0 2026.79  5000.0 2027.97  5005.7 2031.45  5010.9 2028.83  5037.2 2041.31
  5055.3 2053.72  5060.4 2054.55  5110.0 2055.69  5211.0 2055.32  5241.7 2052.94
  5303.2 2054.97  5397.4 2055.76  5486.1 2056.28  5535.7 2058.52  5573.8 2057.59
#Mann=6,-1,0
  4211.4    0.07       0  4266.5   0.035       0  4500.3    0.07       0
  4980.6    0.07       0  4992.0    0.07       0  5397.4   0.045       0
Bank Sta=4980.6,4992
Exp/Cntr=0.3,0.1

Type RM Length L Ch R = 1,91486,420,420,420
BEGIN DESCRIPTION:
Alkali Creek 94.0
END DESCRIPTION:
XS GIS Cut Line= 3
      1347382.92      6953150.02      1348005.00      6953188.00
      1348923.71      6952872.24
#Sta/Elev= 30
  4368.4 2057.97  4380.5 2058.62  4416.4 2055.63  4450.6 2054.87  4490.7 2054.94
  4500.7 2056.48  4553.1 2054.88  4711.1 2053.14  4951.6 2053.87  4981.6 2051.67
  4989.1 2040.68  4994.3 2040.68  5002.0 2032.49  5007.3 2032.83  5017.7 2026.15
  5018.2 2025.65  5029.1 2026.15  5033.2 2028.81  5038.5 2028.19  5069.7 2031.41
  5095.7 2035.88  5245.4 2047.21  5297.3 2049.12  5308.8 2049.72  5376.9 2053.64
  5546.0 2053.72  5676.5 2054.03  5772.5 2054.79  5853.5 2054.64  5963.1 2054.79
#Mann=10,-1,0
  4368.4   0.045       0  4553.1    0.07       0  5017.7    0.07       0
  5029.1    0.07       0  5297.3   0.035       0  5308.8    0.07       0
  5546.0   0.035       0  5676.5    0.07       0  5772.5   0.035       0
  5853.5   0.045       0
Bank Sta=5017.7,5029.1
Exp/Cntr=0.3,0.1

Type RM Length L Ch R = 1,91066,458,458,458
BEGIN DESCRIPTION:
Alkali Creek 93.0
END DESCRIPTION:
XS GIS Cut Line= 3
      1347632.50      6953377.89      1348255.00      6953488.00
      1348728.38      6953536.31
#Sta/Elev= 30
  4367.4 2053.31  4401.1 2053.72  4522.3 2052.05  4568.5 2053.59  4573.5 2052.79
  4627.6 2051.88  4660.8 2052.08  4725.4 2051.30  4766.0 2046.47  4800.1 2045.48
  4844.7 2042.06  4877.7 2038.80  4913.3 2033.01  4918.4 2034.30  4948.8 2030.59
  4979.3 2029.15  4983.5 2025.35  4984.0 2024.85  4995.3 2025.35  4997.0 2028.31
  5021.2 2030.73  5029.7 2033.11  5046.8 2050.53  5051.8 2051.20  5069.9 2049.44
  5110.1 2051.47  5175.3 2051.93  5381.8 2052.23  5451.4 2052.30  5475.4 2052.47
#Mann=9,-1,0
  4367.4    0.07       0  4660.8   0.035       0  4844.7    0.07       0
  4983.5    0.07       0  4995.3    0.07       0  5021.2   0.035       0
  5175.3    0.07       0  5381.8   0.035       0  5451.4    0.07       0
Bank Sta=4983.5,4995.3
Exp/Cntr=0.3,0.1

Type RM Length L Ch R = 1,90608,442,442,442
BEGIN DESCRIPTION:
Alkali Creek 92.0
END DESCRIPTION:
XS GIS Cut Line= 3
      1347829.95      6953913.00      1348105.00      6953888.00
      1348706.67      6953807.58
#Sta/Elev= 30
  4720.1 2051.08  4755.3 2051.90  4865.7 2050.80  4905.9 2051.95  4936.0 2049.77
  4946.1 2048.58  4956.1 2037.80  4966.2 2031.18  4970.2 2024.42  4970.7 2023.92
  4982.2 2024.42  4993.8 2028.01  5006.4 2028.44  5013.1 2027.79  5037.8 2028.00
  5056.8 2029.58  5066.9 2030.55  5077.0 2033.83  5113.5 2036.19  5129.0 2037.48
  5167.8 2039.23  5177.9 2040.94  5208.1 2042.96  5314.1 2047.92  5329.2 2048.43
  5340.1 2050.32  5349.4 2050.70  5486.2 2049.85  5520.9 2051.11  5603.3 2051.19
#Mann=7,-1,0
  4720.1    0.07       0  4970.2    0.07       0  4982.2    0.07       0
  5013.1   0.035       0  5113.5    0.07       0  5129.0   0.035       0
  5314.1    0.07       0
Bank Sta=4970.2,4982.2
Exp/Cntr=0.3,0.1

Type RM Length L Ch R = 1,90166,469,469,469
BEGIN DESCRIPTION:
Alkali Creek 91.0
END DESCRIPTION:
XS GIS Cut Line= 3
      1348030.01      6954362.99      1348405.00      6954188.00
      1348836.88      6953974.68
#Sta/Elev= 30
  4585.7 2049.66  4684.1 2049.35  4802.5 2048.14  4819.8 2046.35  4834.0 2043.27
  4842.7 2043.48  4848.2 2039.80  4865.5 2039.19  4871.0 2036.62  4888.4 2034.59
  4900.2 2031.85  4939.6 2027.47  4955.4 2027.29  4977.4 2025.18  4979.3 2022.53
  4979.8 2022.03  4991.3 2022.53  4996.8 2027.28  5002.3 2027.28  5021.8 2036.96
  5036.0 2037.78  5052.8 2036.80  5066.4 2037.92  5097.7 2041.87  5111.0 2045.29
  5133.3 2047.65  5155.7 2049.06  5203.8 2048.59  5222.6 2049.71  5481.2 2050.34
#Mann=5,-1,0
  4585.7    0.07       0  4684.1   0.035       0  4979.3   0.035       0
  4991.3   0.035       0  5203.8    0.07       0
Bank Sta=4979.3,4991.3
Exp/Cntr=0.3,0.1

Type RM Length L Ch R = 1,89697,422,422,422
BEGIN DESCRIPTION:
Alkali Creek 90.0
END DESCRIPTION:
XS GIS Cut Line= 3
      1348229.96      6954563.00      1348655.00      6954538.00
      1349145.05      6954391.34
#Sta/Elev= 30
  4573.7 2048.05  4608.8 2048.45  4628.8 2047.33  4678.9 2046.66  4769.1 2041.13
  4829.2 2038.37  4868.4 2035.57  4899.3 2033.62  4909.3 2033.70  4920.8 2031.71
  4959.4 2026.47  4969.4 2026.67  4979.4 2024.83  4990.9 2021.50  4991.4 2021.00
  5003.0 2021.50  5009.9 2024.70  5016.0 2026.46  5021.2 2029.61  5030.8 2033.85
  5041.2 2036.63  5049.1 2042.93  5054.3 2041.34  5062.1 2044.49  5072.5 2045.75
  5087.4 2045.61  5135.2 2048.13  5186.7 2047.52  5323.1 2048.42  5511.0 2048.52
#Mann=5,-1,0
  4573.7    0.07       0  4868.4   0.035       0  4920.8    0.07       0
  4990.9    0.07       0  5003.0    0.07       0
Bank Sta=4990.9,5003
Exp/Cntr=0.3,0.1

Type RM Length L Ch R = 1,89275,482,482,482
BEGIN DESCRIPTION:
Alkali Creek 89.0
END DESCRIPTION:
XS GIS Cut Line= 3
      1348079.96      6954812.99      1348655.00      6954888.00
      1349055.60      6954858.50
#Sta/Elev= 30
  4424.9 2047.10  4530.8 2046.53  4571.2 2046.95  4601.4 2046.07  4702.3 2045.22
  4712.4 2045.53  4782.9 2042.98  4873.7 2038.09  4883.8 2036.62  4924.1 2033.57
  4944.3 2031.39  4962.8 2028.20  4974.6 2025.03  4984.6 2023.83  4996.2 2020.91
  4996.7 2020.41  5007.8 2020.41  5008.3 2020.91  5024.9 2024.77  5034.9 2025.22
  5071.4 2031.51  5076.5 2031.31  5085.0 2036.39  5095.1 2040.00  5105.1 2040.45
  5135.2 2044.23  5145.2 2044.79  5228.0 2045.01  5348.0 2045.21  5406.5 2044.29
#Mann=4,-1,0
  4424.9    0.07       0  4996.2   0.035       0  5008.3    0.07       0
  5228.0    0.07       0
Bank Sta=4996.2,5008.3
Exp/Cntr=0.3,0.1

Type RM Length L Ch R = 1,88793,456,456,456
BEGIN DESCRIPTION:
Alkali Creek 88.0
END DESCRIPTION:
XS GIS Cut Line= 3
      1348330.00      6955363.00      1348555.00      6955338.00
      1349002.11      6955001.96
#Sta/Elev= 30
  4774.6 2040.71  4819.9 2041.17  4890.3 2040.05  4970.8 2037.43  4980.9 2036.12
  4990.9 2030.77  4998.5 2025.30  5004.1 2025.30  5008.3 2021.15  5014.5 2021.30
  5023.1 2019.28  5023.6 2018.78  5035.2 2019.28  5037.4 2023.26  5043.7 2022.97
  5051.0 2024.20  5079.1 2024.68  5122.8 2028.06  5201.1 2032.20  5258.2 2036.19
  5293.6 2036.55  5308.2 2037.77  5322.8 2037.48  5337.3 2038.62  5343.6 2037.93
  5367.8 2038.53  5508.1 2039.18  5522.7 2039.40  5529.0 2040.31  5560.3 2039.90
#Mann=5,-1,0
  4774.6    0.07       0  5023.1    0.07       0  5035.2    0.07       0
  5201.1   0.035       0  5367.8    0.07       0
Bank Sta=5023.1,5035.2
Exp/Cntr=0.3,0.1

Type RM Length L Ch R = 1,88337,445,445,445
BEGIN DESCRIPTION:
Alkali Creek 87.0
END DESCRIPTION:
XS GIS Cut Line= 5
      1348430.03      6955613.00      1348862.94      6955531.77
      1348955.00      6955438.00      1349053.91      6955370.31
      1349537.07      6955262.84
#Sta/Elev= 30
  4432.2 2039.17  4738.5 2038.75  4810.2 2036.43  4815.3 2033.98  4823.9 2033.35
  4834.1 2030.61  4867.8 2027.67  4871.2 2026.00  4886.3 2025.22  4933.4 2022.92
  4940.4 2023.45  4976.7 2019.10  4977.2 2018.60  4989.0 2019.10  5007.1 2020.29
  5011.5 2022.10  5017.6 2021.43  5026.4 2024.16  5032.5 2024.65  5040.4 2027.36
  5047.4 2031.20  5053.5 2030.78  5083.3 2034.81  5104.3 2034.09  5135.3 2036.23
  5196.8 2037.48  5300.0 2035.24  5463.1 2035.60  5514.3 2036.22  5618.9 2039.94
#Mann=5,-1,0
  4432.2    0.07       0  4738.5   0.035       0  4886.3    0.07       0
  4976.7    0.07       0  4989.0    0.07       0
Bank Sta=4976.7,4989
Exp/Cntr=0.3,0.1

Type RM Length L Ch R = 1,87892,857,857,857
BEGIN DESCRIPTION:
Alkali Creek 86.0
END DESCRIPTION:
XS GIS Cut Line= 3
      1348613.40      6955783.50      1349155.00      6955788.00
      1349455.05      6955737.99
#Sta/Elev= 30
  4457.8 2037.53  4568.5 2037.29  4619.4 2036.82  4639.4 2035.78  4649.4 2036.17
  4679.4 2035.15  4789.4 2029.98  4829.4 2026.60  4849.4 2027.21  4899.4 2027.27
  4929.4 2025.51  4939.4 2024.01  4959.4 2022.46  4969.4 2022.40  4989.4 2020.59
  5019.7 2019.98  5026.2 2017.86  5026.7 2017.36  5038.1 2017.36  5038.6 2017.86
  5040.0 2021.23  5050.1 2025.81  5070.4 2028.06  5093.2 2027.38  5121.1 2029.14
  5161.6 2029.68  5226.4 2032.13  5270.6 2034.88  5275.7 2034.46  5303.6 2035.96
#Mann=5,-1,0
  4457.8   0.035       0  4568.5    0.07       0  5026.2    0.07       0
  5038.6    0.07       0  5226.4   0.035       0
Bank Sta=5026.2,5038.6
Exp/Cntr=0.3,0.1

Type RM Length L Ch R = 1,87035,617,617,617
BEGIN DESCRIPTION:
Alkali Creek 85.0
END DESCRIPTION:
XS GIS Cut Line= 3
      1348329.97      6956012.99      1348955.00      6956238.00
      1349680.03      6956163.00
#Sta/Elev= 30
  4341.8 2036.25  4513.7 2035.95  4598.7 2035.11  4708.5 2034.90  4787.3 2033.23
  4825.4 2033.29  4891.5 2031.26  4903.9 2030.12  4921.1 2018.57  4929.3 2015.22
  4934.7 2019.15  4942.3 2016.58  4965.4 2018.64  4974.2 2017.81  4978.6 2014.76
  4979.1 2014.26  4991.0 2014.76  5003.4 2019.40  5026.2 2021.26  5058.0 2027.21
  5156.9 2030.49  5227.3 2031.04  5276.9 2030.26  5438.4 2033.11  5461.1 2035.02
  5508.8 2033.21  5589.2 2034.22  5641.1 2036.53  5669.6 2035.31  5735.0 2037.26
#Mann=9,-1,0
  4341.8    0.07       0  4513.7   0.035       0  4598.7    0.07       0
  4787.3   0.035       0  4891.5    0.07       0  4978.6    0.07       0
  4991.0    0.07       0  5276.9   0.035       0  5461.1   0.045       0
Bank Sta=4978.6,4991
Exp/Cntr=0.3,0.1

Type RM Length L Ch R = 1,86418,463,463,463
BEGIN DESCRIPTION:
Alkali Creek 84.0
END DESCRIPTION:
XS GIS Cut Line= 3
      1348812.03      6956430.80      1348903.17      6956769.32
      1348999.51      6956847.43
#Sta/Elev= 30
  4733.5 2029.55  4772.0 2029.25  4834.2 2027.64  4840.2 2026.93  4854.9 2027.16
  4865.2 2030.28  4875.0 2029.80  4880.2 2030.44  4885.9 2028.76  4906.7 2025.13
  4914.9 2024.10  4920.1 2024.95  4948.1 2019.97  4954.9 2017.76  4960.0 2018.41
  4968.8 2016.48  4972.9 2014.28  4973.4 2013.78  4984.9 2013.78  4985.4 2014.28
  4989.5 2017.18  5000.0 2018.40  5029.6 2025.71  5034.8 2025.28  5041.3 2027.43
  5062.0 2029.95  5141.0 2032.12  5176.5 2031.44  5184.1 2032.13  5208.1 2031.02
#Mann=3,-1,0
  4733.5    0.07       0  4972.9    0.07       0  4985.4    0.07       0
Bank Sta=4972.9,4985.4
Exp/Cntr=0.3,0.1

Type RM Length L Ch R = 1,85955,476,476,476
BEGIN DESCRIPTION:
Alkali Creek 83.1
END DESCRIPTION:
XS GIS Cut Line= 3
      1348254.74      6956633.91      1348605.43      6956908.18
      1348980.09      6956892.22
#Sta/Elev= 30
  4554.8 2032.20  4615.3 2032.45  4636.1 2031.42  4662.1 2031.69  4671.3 2031.11
  4814.2 2031.05  4892.9 2028.86  4913.7 2027.68  4942.6 2023.99  4949.0 2024.99
  4957.1 2022.76  4963.4 2021.88  4971.5 2018.83  4978.8 2018.39  4986.0 2017.66
  4990.3 2013.84  4990.8 2013.34  5002.8 2013.84  5029.6 2018.43  5039.6 2022.24
  5049.6 2023.50  5059.6 2022.61  5069.6 2023.27  5089.7 2026.00  5118.2 2027.10
  5139.7 2026.98  5189.7 2029.55  5219.8 2030.31  5289.8 2031.26  5375.0 2030.93
#Mann=5,-1,0
  4554.8    0.07       0  4662.1   0.035       0  4978.8    0.07       0
  4990.3    0.07       0  5002.8    0.07       0
Bank Sta=4990.3,5002.8
Exp/Cntr=0.3,0.1

Type RM Length L Ch R = 1,85479,265,265,265
BEGIN DESCRIPTION:
Alkali Creek 83.2
END DESCRIPTION:
XS GIS Cut Line= 2
      1348072.41      6957706.84      1348884.95      6956964.63
#Sta/Elev= 30
  4397.5 2031.17  4490.6 2030.30  4525.7 2031.00  4554.1 2030.34  4589.9 2031.02
  4639.2 2030.35  4653.4 2030.97  4710.2 2030.07  4731.1 2031.07  4780.4 2029.13
  4851.4 2028.52  4873.0 2027.19  4943.3 2026.10  4957.4 2024.14  4970.3 2011.85
  4970.8 2011.35  4987.3 2011.35  4987.8 2011.85  4993.2 2015.25  5028.4 2017.55
  5070.9 2019.12  5085.1 2020.67  5106.1 2021.26  5141.9 2025.33  5162.8 2025.66
  5184.4 2027.28  5254.7 2027.89  5268.9 2027.34  5396.6 2030.06  5498.0 2030.76
#Mann=3,-1,0
  4397.5    0.07       0  4970.3    0.07       0  4987.8    0.07       0
Bank Sta=4970.3,4987.8
Exp/Cntr=0.3,0.1

Type RM Length L Ch R = 1,85214,1321,1321,1321
BEGIN DESCRIPTION:
Alkali Creek 83.0
END DESCRIPTION:
XS GIS Cut Line= 3
      1348265.13      6957855.27      1348705.00      6957488.00
      1349170.23      6957093.22
#Sta/Elev= 30
  4426.7 2030.36  4574.0 2029.88  4659.4 2030.15  4723.2 2028.76  4772.6 2026.19
  4815.6 2022.47  4822.1 2023.06  4836.4 2022.16  4850.7 2019.92  4871.6 2020.68
  4900.2 2020.07  4964.0 2017.01  4992.6 2014.74  4996.5 2012.86  4998.1 2010.35
  4998.6 2009.85  5015.6 2010.35  5021.2 2014.52  5027.7 2014.54  5035.5 2022.14
  5056.3 2025.57  5205.7 2025.83  5234.3 2024.36  5240.8 2025.25  5248.6 2024.06
  5255.1 2025.09  5298.0 2026.69  5414.0 2027.44  5540.2 2028.65  5609.9 2029.16
#Mann=6,-1,0
  4426.7   0.035       0  4574.0    0.07       0  4998.1    0.07       0
  5015.6    0.07       0  5414.0   0.035       0  5540.2    0.07       0
Bank Sta=4998.1,5015.6
Exp/Cntr=0.3,0.1

Type RM Length L Ch R = 1,83893,487,487,487
BEGIN DESCRIPTION:
Alkali Creek 82.0
END DESCRIPTION:
XS GIS Cut Line= 3
      1348304.99      6958038.00      1349405.00      6957538.00
      1350405.02      6956337.97
#Sta/Elev= 30
  3791.2 2031.67  3985.9 2029.97  4208.6 2027.92  4219.6 2021.16  4237.2 2028.54
  4242.7 2024.50  4260.3 2027.58  4265.7 2022.38  4283.3 2025.82  4288.8 2018.76
  4306.4 2022.77  4311.9 2017.52  4329.5 2024.84  4340.4 2022.31  4363.5 2022.86
  4381.1 2027.33  4442.6 2026.94  4823.8 2021.59  4985.2 2013.13  4997.9 2009.62
  4998.4 2009.12  5015.4 2009.62  5021.0 2019.09  5035.3 2022.47  5171.6 2024.98
  5255.3 2027.66  5350.4 2025.46  5820.4 2028.50  6149.6 2033.13  6561.6 2047.02
#Mann=8,-1,0
  3791.2   0.063       0  3985.9   0.035       0  4442.6    0.07       0
  4997.9    0.07       0  5015.4    0.07       0  5171.6   0.035       0
  5350.4    0.07       0  5820.4   0.045       0
Bank Sta=4997.9,5015.4
Exp/Cntr=0.3,0.1

Type RM Length L Ch R = 1,83406,138,138,138
BEGIN DESCRIPTION:
Alkali Creek 81.0
END DESCRIPTION:
XS GIS Cut Line= 4
      1348598.56      6957965.98      1348973.61      6957965.98
      1349484.46      6957967.85      1349931.86      6957968.14
#Sta/Elev= 30
  4114.1 2029.73  4290.5 2028.42  4360.5 2026.52  4560.5 2023.70  4720.5 2023.70
  4870.5 2022.93  4900.5 2021.96  4910.5 2022.42  4930.5 2020.81  4940.5 2017.13
  4950.5 2016.51  4980.5 2012.34  4981.7 2011.22  4982.2 2010.72  4998.9 2010.72
  4999.4 2011.22  5030.5 2012.66  5060.5 2012.90  5100.5 2015.73  5110.5 2014.98
  5120.5 2015.87  5130.5 2018.84  5140.5 2020.53  5170.5 2023.71  5190.5 2023.77
  5200.5 2022.93  5220.5 2024.29  5290.5 2025.74  5370.5 2024.80  5447.4 2025.35
#Mann=3,-1,0
  4114.1   0.035       0  4981.7   0.035       0  4999.4   0.035       0
Bank Sta=4981.7,4999.4
Exp/Cntr=0.3,0.1

Type RM Length L Ch R = 1,83268,1174,1174,1174
BEGIN DESCRIPTION:
Alkali Creek 80.5
END DESCRIPTION:
XS GIS Cut Line= 2
      1348588.15      6958077.38      1349990.43      6958111.43
#Sta/Elev= 30
  4082.8 2030.04  4089.7 2029.19  4269.7 2028.49  4279.7 2027.50  4314.6 2027.61
  4329.7 2026.07  4449.8 2023.88  4519.8 2023.23  4689.8 2023.44  4879.9 2021.52
  4895.7 2020.75  4919.9 2019.81  4929.9 2016.67  4949.9 2013.20  4959.9 2011.91
  4979.9 2011.24  4981.1 2010.37  4981.6 2009.87  4998.3 2009.87  4998.8 2010.37
  5039.9 2016.52  5059.9 2022.18  5069.9 2024.17  5120.0 2025.90  5170.0 2025.04
  5219.8 2025.46  5310.0 2025.73  5330.0 2025.12  5460.1 2025.22  5485.5 2024.63
#Mann=5,-1,0
  4082.8   0.035       0  4895.7   0.063       0  4981.1   0.063       0
  4998.8   0.063       0  5219.8   0.035       0
Bank Sta=4981.1,4998.8
Exp/Cntr=0.3,0.1

Type RM Length L Ch R = 1,82094,1372,1372,1372
BEGIN DESCRIPTION:
Alkali Creek 80.0
END DESCRIPTION:
XS GIS Cut Line= 4
      1347977.19      6959359.43      1349005.00      6958638.00
      1349654.24      6958416.75      1351204.98      6957438.02
#Sta/Elev= 30
  3749.9 2039.50  4504.1 2029.50  4796.3 2028.15  4855.3 2027.43  4926.8 2022.16
  4941.6 2020.19  4947.7 2016.33  4956.4 2017.46  4962.5 2012.34  4989.1 2008.21
  4989.6 2007.71  5007.3 2008.21  5052.7 2013.82  5121.8 2017.54  5298.1 2016.90
  5608.0 2024.22  5776.7 2024.30  6011.5 2024.59  6271.9 2025.03  6315.1 2022.48
  6388.0 2024.84  6451.6 2022.18  6509.2 2025.36  6763.9 2023.79  6899.0 2024.17
  7299.7 2026.05  7430.7 2028.56  7475.3 2026.26  7496.5 2029.52  7525.3 2028.50
#Mann=10,-1,0
  3749.9   0.035       0  4796.3    0.07       0  4989.1    0.07       0
  5007.3    0.07       0  5608.0   0.035       0  5776.7    0.07       0
  6011.5   0.035       0  6763.9    0.07       0  6899.0   0.045       0
  7299.7   0.035       0
Bank Sta=4989.1,5007.3
Exp/Cntr=0.3,0.1

Type RM Length L Ch R = 1,80722,476,476,476
BEGIN DESCRIPTION:
Alkali Creek 79.0
END DESCRIPTION:
XS GIS Cut Line= 3
      1348805.01      6959188.00      1349805.00      6959088.00
      1352205.01      6956687.99
#Sta/Elev= 30
  3994.9 2030.69  4223.6 2025.80  4478.8 2021.05  4607.9 2019.03  4708.4 2013.44
  4768.7 2014.11  4819.0 2008.47  4947.1 2008.40  4969.7 2010.75  5003.4 2010.39
  5019.1 2007.30  5019.6 2006.80  5037.3 2007.30  5056.4 2009.39  5070.6 2019.34
  5098.9 2021.27  5379.4 2021.51  5440.4 2022.19  6180.6 2022.19  6371.7 2019.29
  6456.5 2025.52  6513.1 2022.81  6555.5 2026.70  6640.4 2024.44  6810.1 2024.83
  6838.4 2028.33  6943.0 2026.97  7333.3 2027.72  7658.6 2031.94  8394.0 2058.79
#Mann=9,-1,0
  3994.9    0.07       0  4223.6   0.035       0  4478.8    0.07       0
  5019.1    0.07       0  5037.3    0.07       0  5379.4   0.035       0
  5440.4    0.07       0  6180.6   0.035       0  6943.0   0.045       0
Bank Sta=5019.1,5037.3
Exp/Cntr=0.3,0.1

Type RM Length L Ch R = 1,80246,472,472,472
BEGIN DESCRIPTION:
Alkali Creek 78.0
END DESCRIPTION:
XS GIS Cut Line= 3
      1349229.31      6960207.14      1349605.00      6959488.00
      1352005.02      6957087.98
#Sta/Elev= 30
  4184.4 2050.66  4648.1 2038.78  4730.3 2035.25  4804.0 2030.58  4810.9 2023.72
  4816.5 2030.84  4833.0 2026.08  4838.6 2029.59  4855.1 2019.08  4881.7 2017.09
  4959.8 2011.37  4978.2 2007.50  4978.7 2007.00  4996.8 2007.50  5207.9 2015.58
  5504.9 2020.16  6739.4 2021.51  6890.8 2021.86  7003.9 2025.74  7074.6 2023.01
  7117.1 2026.44  7222.0 2024.58  7244.4 2023.95  7258.5 2027.18  7286.8 2027.44
  7456.5 2026.12  7951.5 2029.34  8135.3 2034.11  8333.3 2043.50  8389.9 2043.78
#Mann=8,-1,0
  4184.4   0.035       0  4648.1    0.07       0  4730.3   0.035       0
  4881.7    0.07       0  4978.2    0.07       0  4996.8    0.07       0
  6739.4   0.035       0  7222.0   0.045       0
Bank Sta=4978.2,4996.8
Exp/Cntr=0.3,0.1

Type RM Length L Ch R = 1,79774,479,479,479
BEGIN DESCRIPTION:
Alkali Creek 77.0
END DESCRIPTION:
XS GIS Cut Line= 3
      1349392.07      6960337.34      1350005.00      6959538.00
      1352204.97      6957138.04
#Sta/Elev= 30
  3992.6 2050.75  4151.3 2048.84  4614.6 2029.91  4749.7 2015.11  4807.2 2012.33
  4927.9 2008.96  4947.9 2006.50  4948.4 2006.00  4966.6 2006.50  5381.9 2019.13
  6719.4 2022.40  6735.7 2022.23  6896.9 2021.37  6917.9 2024.07  6939.5 2021.49
  6974.6 2025.85  7045.5 2023.54  7137.4 2027.38  7205.7 2025.98  7682.5 2029.48
  7880.4 2037.97  7923.0 2037.26  7958.1 2040.53  8008.1 2039.89  8043.2 2043.74
  8106.7 2043.94  8142.5 2047.36  8177.6 2046.27  8220.2 2050.22  8255.6 2049.63
#Mann=9,-1,0
  3992.6    0.07       0  4151.3   0.035       0  4807.2    0.16       0
  4927.9    0.07       0  4947.9    0.07       0  4966.6    0.07       0
  6719.4   0.045       0  6735.7   0.035       0  7205.7   0.045       0
Bank Sta=4947.9,4966.6
Exp/Cntr=0.3,0.1

Type RM Length L Ch R = 1,79295,471,471,471
BEGIN DESCRIPTION:
Alkali Creek 76.0
END DESCRIPTION:
XS GIS Cut Line= 3
      1349576.52      6960586.92      1350455.00      6959538.00
      1351805.00      6957738.00
#Sta/Elev= 30
  3636.4 2043.19  3693.1 2039.87  3748.4 2041.34  4057.8 2036.77  4429.1 2029.44
  4471.6 2027.68  4699.0 2019.14  4906.5 2010.24  4992.0 2007.54  4992.5 2007.04
  5010.7 2007.54  5076.5 2014.43  5147.1 2015.62  5282.7 2018.31  5911.9 2018.40
  6091.1 2021.94  6118.1 2018.76  6211.9 2024.14  6218.1 2021.00  6274.8 2020.78
  6526.5 2019.87  6600.8 2022.00  6747.3 2021.47  6768.1 2025.03  6791.1 2023.52
  6847.3 2026.48  6897.3 2023.99  6954.6 2027.93  7038.5 2025.83  7254.6 2027.89
#Mann=13,-1,0
  3636.4   0.045       0  3693.1    0.07       0  4057.8   0.035       0
  4429.1    0.07       0  4471.6   0.035       0  4699.0    0.07       0
  4906.5    0.16       0  4992.0    0.07       0  5010.7    0.16       0
  5147.1    0.07       0  6274.8   0.045       0  6600.8   0.035       0
  7038.5   0.045       0
Bank Sta=4992,5010.7
Exp/Cntr=0.3,0.1

Type RM Length L Ch R = 1,78824,466,466,466
BEGIN DESCRIPTION:
Alkali Creek 75.0
END DESCRIPTION:
XS GIS Cut Line= 3
      1349826.11      6960901.56      1350855.00      6959738.00
      1352255.00      6957338.01
#Sta/Elev= 30
  3446.9 2038.43  3727.5 2033.12  3751.3 2033.05  4490.3 2023.42  4653.1 2019.13
  4780.5 2012.38  5137.5 2010.33  5138.0 2009.83  5156.3 2010.33  5174.2 2014.06
  5584.1 2015.60  5949.4 2016.19  5995.7 2018.57  6541.9 2018.15  6706.1 2020.84
  6841.3 2021.74  6864.0 2025.21  6878.5 2023.69  6921.9 2027.05  6968.2 2024.79
  7117.0 2028.23  7215.1 2032.01  7252.3 2030.65  7316.8 2035.11  7348.2 2033.79
  7397.0 2037.78  7449.9 2036.63  7492.9 2040.55  7545.8 2039.42  7778.6 2044.65
#Mann=8,-1,0
  3446.9   0.045       0  3727.5   0.035       0  3751.3    0.07       0
  5137.5    0.07       0  5156.3    0.07       0  5584.1   0.045       0
  6706.1   0.035       0  7117.0   0.045       0
Bank Sta=5137.5,5156.3
Exp/Cntr=0.3,0.1

Type RM Length L Ch R = 1,78358,445,445,445
BEGIN DESCRIPTION:
Alkali Creek 74.0
END DESCRIPTION:
XS GIS Cut Line= 3
      1350305.01      6960987.99      1351305.00      6959788.00
      1352495.40      6957635.47
#Sta/Elev= 30
  3437.6 2036.07  3473.4 2032.51  3551.5 2033.19  3593.8 2029.53  3699.9 2030.89
  3736.3 2026.63  3800.1 2024.97  3927.7 2026.48  4020.1 2021.92  4225.8 2021.26
  4480.9 2014.20  4807.6 2012.49  4968.8 2007.23  4969.3 2006.73  4987.6 2007.23
  5056.9 2007.44  5115.6 2012.25  5881.5 2012.69  5935.4 2015.31  6353.4 2015.16
  6735.3 2020.20  6890.6 2023.90  6942.3 2027.77  6993.7 2026.60  7009.7 2030.07
  7059.0 2030.85  7090.8 2035.06  7149.1 2035.20  7178.1 2037.51  7459.4 2037.06
#Mann=6,-1,0
  3437.6    0.07       0  4968.8    0.07       0  4987.6    0.07       0
  5115.6   0.045       0  6735.3   0.035       0  7149.1   0.045       0
Bank Sta=4968.8,4987.6
Exp/Cntr=0.3,0.1

Type RM Length L Ch R = 1,77913,907,907,907
BEGIN DESCRIPTION:
Alkali Creek 73.0
END DESCRIPTION:
XS GIS Cut Line= 3
      1350504.97      6961138.03      1351705.00      6959938.00
      1352605.02      6958137.97
#Sta/Elev= 30
  3307.1 2039.25  3434.4 2032.23  3476.9 2033.66  3575.8 2028.41  3618.3 2029.98
  3759.7 2020.95  3887.0 2019.01  3915.3 2020.96  4099.1 2014.15  4226.4 2013.31
  4254.7 2010.48  4480.9 2007.60  4537.5 2010.12  4650.6 2005.63  4763.8 2010.56
  4909.8 2009.80  4991.2 2005.39  4991.7 2004.89  5010.1 2005.39  5138.4 2010.60
  5979.7 2009.78  6063.5 2012.77  6270.4 2012.52  6323.5 2015.12  6516.3 2015.17
  6667.3 2018.96  6784.7 2018.60  6837.8 2021.75  6865.2 2020.37  7016.7 2025.69
#Mann=5,-1,0
  3307.1    0.07       0  4909.8   0.045       0  4991.2   0.045       0
  5010.1   0.045       0  6865.2   0.035       0
Bank Sta=4991.2,5010.1
Exp/Cntr=0.3,0.1

Type RM Length L Ch R = 1,77006,450,450,450
BEGIN DESCRIPTION:
Alkali Creek 72.0
END DESCRIPTION:
XS GIS Cut Line= 3
      1351063.08      6961324.76      1351605.00      6960588.00
      1353416.99      6957831.89
#Sta/Elev= 30
  4081.8 2038.48  4115.8 2039.55  4174.4 2035.28  4209.9 2036.66  4245.4 2032.86
  4338.5 2033.81  4395.8 2030.04  4552.4 2029.09  4577.4 2026.14  4692.7 2023.98
  4732.2 2020.51  4788.5 2020.39  5015.5 2003.06  5016.0 2002.56  5034.5 2003.06
  5061.2 2005.92  5097.3 2004.31  5284.1 2010.85  5354.5 2010.02  5892.7 2007.25
  6468.4 2008.26  7299.6 2016.22  7625.0 2022.61  7758.5 2021.18  7790.7 2023.69
  7905.2 2024.15  7964.4 2030.06  8043.8 2027.42  8211.9 2030.41  8294.8 2031.76
#Mann=8,-1,0
  4081.8    0.07       0  4577.4   0.035       0  4692.7    0.07       0
  5015.5    0.07       0  5034.5    0.07       0  5354.5   0.045       0
  7758.5   0.035       0  8211.9   0.045       0
Bank Sta=5015.5,5034.5
Exp/Cntr=0.3,0.1

Type RM Length L Ch R = 1,76556,454,454,454
BEGIN DESCRIPTION:
Alkali Creek 71.0
END DESCRIPTION:
XS GIS Cut Line= 3
      1351388.63      6961465.78      1352005.00      6960588.00
      1354005.02      6958187.98
#Sta/Elev= 30
  3918.9 2040.82  4058.6 2035.84  4130.1 2037.04  4201.5 2032.36  4237.3 2033.71
  4273.0 2029.83  4344.4 2029.27  4430.7 2022.92  4460.3 2024.15  4502.7 2019.80
  4539.4 2020.83  4582.3 2016.99  4719.1 2014.45  4918.7 2004.27  4994.7 2003.88
  5010.0 2001.35  5010.5 2000.85  5029.0 2001.35  5076.7 2007.93  5113.5 2005.97
  6653.1 2006.07  6844.5 2013.14  6930.4 2012.05  6979.8 2014.96  7022.1 2013.25
  7660.6 2021.33  7984.3 2031.85  8009.5 2034.81  8051.1 2033.48  8115.6 2036.63
#Mann=5,-1,0
  3918.9    0.07       0  5010.0    0.07       0  5029.0    0.07       0
  5113.5   0.045       0  7984.3   0.035       0
Bank Sta=5010,5029
Exp/Cntr=0.3,0.1

Type RM Length L Ch R = 1,76102,469,469,469
BEGIN DESCRIPTION:
Alkali Creek 70.0
END DESCRIPTION:
XS GIS Cut Line= 3
      1351551.36      6961585.16      1352405.00      6960738.00
      1354205.03      6958337.96
#Sta/Elev= 30
  3796.6 2038.70  3882.0 2037.04  3945.6 2032.23  3981.0 2033.28  4023.5 2029.16
  4164.9 2027.04  4200.2 2023.38  4256.8 2024.13  4320.4 2019.58  4348.7 2021.05
  4384.1 2017.14  4483.1 2017.00  4511.3 2013.59  4582.1 2013.18  4666.9 2007.41
  4971.0 2002.78  5012.8 2001.68  5017.9 1999.46  5018.4 1998.96  5036.9 1999.46
  5061.5 2005.10  5471.5 2002.94  5476.7 2002.95  5596.6 2002.95  5971.1 2005.23
  6362.8 2003.88  6592.0 2007.77  6649.3 2011.00  7177.4 2012.69  7999.3 2033.96
#Mann=7,-1,0
  3796.6    0.07       0  5017.9    0.07       0  5036.9    0.07       0
  5061.5   0.045       0  5471.5   0.035       0  5476.7    0.07       0
  5596.6   0.045       0
Bank Sta=5017.9,5036.9
Exp/Cntr=0.3,0.1

Type RM Length L Ch R = 1,75633,3206,3206,3206
BEGIN DESCRIPTION:
Alkali Creek 69.0
END DESCRIPTION:
XS GIS Cut Line= 3
      1351746.72      6961693.63      1352355.00      6961088.00
      1354155.02      6958687.97
#Sta/Elev= 30
  4137.7 2036.61  4352.6 2025.73  4508.2 2024.07  4550.6 2019.74  4593.0 2020.87
  4628.4 2016.76  4720.3 2015.42  4755.7 2011.17  4904.1 2010.71  4967.8 2006.27
  4981.9 2002.55  4983.0 1998.85  4983.5 1998.35  5002.1 1998.85  5009.6 2001.69
  5159.6 2001.97  5282.5 2005.79  5381.6 2003.92  5584.4 2002.77  5753.4 1999.06
  5879.8 2000.42  6023.6 2003.15  6052.4 2004.86  6120.0 2003.42  6451.9 2002.92
  6717.9 2002.79  6938.8 2006.00  6982.5 2008.94  7446.1 2010.45  7996.1 2024.64
#Mann=10,-1,0
  4137.7    0.07       0  4983.0    0.07       0  5002.1    0.07       0
  5381.6   0.045       0  5584.4    0.07       0  5879.8   0.035       0
  6023.6    0.07       0  6052.4   0.035       0  6120.0    0.07       0
  6451.9   0.045       0
Bank Sta=4983,5002.1
Exp/Cntr=0.3,0.1
