HEC-RAS study Alkali Creek.prj: Alkali Creek Base Level Engineering

--- Alkali Creek.g01 (geometry) --- (continued)

Type RM Length L Ch R = 1,31565,1268,1268,1268
BEGIN DESCRIPTION:
Alkali Creek 28.0
END DESCRIPTION:
XS GIS Cut Line= 3
      1376605.01      6970187.97      1378005.00      6967088.00
      1378005.00      6963088.04
#Sta/Elev= 30
  1602.4 1972.32  1714.6 1972.12  2183.9 1955.20  2227.8 1951.72  2546.0 1946.14
  3303.1 1944.88  3456.1 1942.59  3559.6 1937.52  3884.6 1934.60  4286.1 1937.28
  4567.6 1931.06  4959.9 1930.87  4976.6 1928.50  4977.5 1928.00  5013.4 1928.50
  5013.8 1931.10  5053.8 1931.50  5846.6 1931.70  5884.1 1931.75  6093.4 1932.02
  6987.8 1933.01  7188.1 1933.62  7389.4 1935.84  7513.8 1939.54  7573.8 1938.74
  7613.8 1942.20  7653.8 1940.22  8233.8 1941.46  8513.8 1947.21  9003.8 1950.79
#Mann=10,-1,0
  1602.4   0.045       0  4567.6    0.07       0  4976.6    0.07       0
  5013.4    0.07       0  5846.6    0.07       0  5884.1   0.045       0
  6093.4    0.07       0  6987.8   0.045       0  7188.1    0.07       0
  7389.4   0.045       0
Bank Sta=4976.6,5013.4
Exp/Cntr=0.3,0.1

Type RM Length L Ch R = 1,30297,984,984,984
BEGIN DESCRIPTION:
Alkali Creek 27.0
END DESCRIPTION:
XS GIS Cut Line= 3
      1376804.99      6969988.01      1378252.72      6968084.29
      1378480.24      6967683.42
#Sta/Elev= 30
  2609.3 1963.58  2645.7 1963.88  2687.3 1959.75  2730.9 1959.91  2751.8 1956.89
  2851.6 1955.08  2901.5 1951.10  2945.1 1952.17  2995.0 1948.68  3758.2 1942.71
  3843.4 1939.83  3901.6 1940.81  3978.7 1937.31  4051.3 1937.71  4107.5 1934.58
  4151.1 1935.66  4192.8 1932.88  4426.5 1931.71  4606.1 1930.47  4766.8 1929.79
  4928.8 1929.96  4993.3 1928.16  4996.1 1926.15  4997.1 1925.65  5033.5 1926.15
  5036.5 1928.96  5042.7 1929.99  5136.5 1933.99  5413.2 1948.90  5461.9 1950.59
#Mann=8,-1,0
  2609.3   0.045       0  4426.5    0.07       0  4606.1   0.045       0
  4766.8    0.07       0  4996.1    0.07       0  5033.5    0.07       0
  5136.5   0.035       0  5413.2    0.07       0
Bank Sta=4996.1,5033.5
Exp/Cntr=0.3,0.1

Type RM Length L Ch R = 1,29313,535,535,535
BEGIN DESCRIPTION:
Alkali Creek 26.0
END DESCRIPTION:
XS GIS Cut Line= 3
      1379254.98      6968637.99      1378805.00      6968338.00
      1378505.00      6967688.00
#Sta/Elev= 30
  4467.6 1950.39  4532.2 1946.41  4562.2 1947.54  4589.3 1945.03  4632.1 1944.74
  4676.4 1943.79  4691.4 1941.57  4742.5 1942.20  4769.5 1939.06  4820.6 1936.80
  4877.7 1931.50  4979.9 1928.24  4985.9 1927.42  4986.6 1925.25  4987.5 1924.75
  5024.3 1925.25  5030.4 1928.87  5074.5 1929.17  5119.9 1927.80  5188.8 1928.86
  5349.4 1936.99  5371.9 1939.30  5446.7 1941.24  5464.3 1942.70  5549.5 1945.36
  5566.9 1947.41  5572.4 1946.36  5595.3 1946.42  5680.7 1948.64  5724.3 1950.43
#Mann=6,-1,0
  4467.6   0.045       0  4632.1    0.07       0  4986.6    0.07       0
  5024.3    0.07       0  5464.3   0.035       0  5680.7    0.07       0
Bank Sta=4986.6,5024.3
Exp/Cntr=0.3,0.1

Type RM Length L Ch R = 1,28778,683,683,683
BEGIN DESCRIPTION:
Alkali Creek 25.0
END DESCRIPTION:
XS GIS Cut Line= 3
      1379455.01      6968438.01      1379155.00      6967988.00
      1378654.97      6967587.98
#Sta/Elev= 30
  4464.1 1952.88  4525.2 1949.88  4615.9 1943.81  4651.9 1942.60  4680.4 1939.75
  4716.5 1937.68  4730.0 1935.67  4745.0 1935.68  4781.1 1932.44  4824.7 1930.07
  4940.3 1928.32  4942.5 1925.05  4943.5 1924.55  4980.2 1925.05  4982.4 1927.11
  5008.2 1926.40  5018.6 1927.89  5097.0 1927.76  5111.4 1928.74  5119.4 1928.10
  5169.0 1930.22  5197.0 1930.41  5381.9 1938.69  5417.2 1941.66  5446.0 1942.20
  5467.9 1943.79  5489.2 1945.19  5559.6 1947.02  5581.2 1949.11  5645.3 1951.43
#Mann=5,-1,0
  4464.1   0.035       0  4525.2    0.07       0  4942.5    0.07       0
  4980.2    0.07       0  5467.9   0.035       0
Bank Sta=4942.5,4980.2
Exp/Cntr=0.3,0.1

Type RM Length L Ch R = 1,28095,28,28,28
BEGIN DESCRIPTION:
Alkali Creek 24.0
END DESCRIPTION:
XS GIS Cut Line= 4
      1379476.53      6968403.43      1379656.43      6967648.69
      1379718.44      6967329.31      1379240.22      6966735.96
#Sta/Elev= 30
  4164.6 1951.94  4219.6 1949.90  4224.7 1947.29  4303.8 1947.12  4351.1 1943.45
  4356.2 1940.70  4393.2 1939.24  4406.6 1935.90  4435.3 1936.34  4447.7 1933.06
  4477.5 1935.05  4488.9 1931.95  4566.8 1932.90  4581.4 1929.77  4609.0 1931.48
  4663.6 1928.88  4943.4 1929.00  4951.4 1928.56  4957.8 1923.07  4962.9 1923.88
  4963.1 1922.09  4964.0 1921.59  5000.8 1922.09  5009.5 1926.95  5022.7 1927.77
  5367.9 1926.18  5617.3 1929.65  5793.5 1935.17  5933.4 1942.49  6027.9 1949.20
#Mann=6,-1,0
  4164.6   0.035       0  4963.1   0.035       0  5000.8   0.035       0
  5367.9    0.07       0  5793.5   0.035       0  5933.4    0.07       0
Bank Sta=4963.1,5000.8
Exp/Cntr=0.3,0.1

Type RM Length L Ch R = 1,28067,1555,1555,1555
BEGIN DESCRIPTION:
Alkali Creek 23.5
END DESCRIPTION:
XS GIS Cut Line= 3
      1379509.41      6968406.96      1379775.02      6967235.12
      1379364.18      6966742.26
#Sta/Elev= 30
  4158.3 1949.53  4161.7 1952.98  4204.8 1948.08  4209.9 1951.27  4247.9 1946.73
  4253.0 1949.21  4382.4 1938.06  4387.6 1941.42  4430.7 1934.47  4435.8 1938.37
  4473.8 1932.71  4478.9 1935.17  4495.6 1935.24  4522.1 1931.21  4527.2 1934.42
  4565.2 1930.59  4570.3 1932.52  4661.7 1928.50  4946.8 1928.45  4968.9 1923.30
  4969.9 1922.80  5006.6 1923.30  5008.3 1926.97  5016.9 1927.91  5339.3 1925.03
  5507.3 1928.03  5698.4 1929.54  5828.3 1934.08  5970.6 1940.33  6001.5 1942.87
#Mann=6,-1,0
  4158.3   0.035       0  4968.9   0.035       0  5006.6   0.035       0
  5507.3    0.07       0  5828.3   0.035       0  5970.6    0.07       0
Bank Sta=4968.9,5006.6
Exp/Cntr=0.3,0.1

Type RM Length L Ch R = 1,26512,541,541,541
BEGIN DESCRIPTION:
Alkali Creek 23.0
END DESCRIPTION:
XS GIS Cut Line= 5
      1379559.39      6968613.50      1380825.07      6967121.69
      1380905.00      6966938.00      1380944.86      6966835.23
      1379455.02      6965638.02
#Sta/Elev= 30
  2847.8 1952.77  2898.0 1952.22  3004.6 1943.50  3047.4 1942.96  3082.6 1938.84
  3111.1 1939.85  3146.2 1935.82  3189.1 1935.75  3238.5 1931.30  3287.9 1931.83
  3316.5 1929.24  3437.3 1926.94  4966.6 1924.70  4971.2 1920.85  4972.1 1920.35
  5009.0 1920.85  5019.5 1923.94  5148.4 1925.10  5817.2 1925.71  6238.5 1927.93
  6321.2 1928.67  6335.6 1931.71  6432.3 1933.67  6492.4 1935.52  6713.2 1947.69
  6748.4 1947.78  6806.0 1950.70  6926.6 1951.80  7001.8 1955.13  7026.0 1955.34
#Mann=7,-1,0
  2847.8   0.045       0  4971.2   0.045       0  5009.0   0.045       0
  6238.5   0.035       0  6432.3    0.07       0  6926.6    0.16       0
  7001.8    0.07       0
Bank Sta=4971.2,5009
Exp/Cntr=0.3,0.1

Type RM Length L Ch R = 1,25971,1604,1604,1604
BEGIN DESCRIPTION:
Alkali Creek 22.0
END DESCRIPTION:
XS GIS Cut Line= 5
      1379555.02      6968687.98      1381332.36      6967210.92
      1381355.00      6967088.00      1381367.08      6966908.84
      1379655.01      6963888.01
#Sta/Elev= 30
  2563.7 1953.99  2641.7 1952.74  2797.7 1939.50  2833.8 1939.87  2883.3 1935.32
  2918.5 1936.22  2961.4 1931.72  3238.8 1926.34  4979.3 1924.79  4989.5 1923.85
  4990.7 1921.68  4991.7 1921.18  5028.6 1921.68  5029.7 1923.81  5059.8 1924.15
  6750.8 1926.67  6893.9 1927.62  7291.4 1930.32  7528.9 1931.49  7565.9 1933.59
  7668.3 1932.87  7733.2 1936.06  7926.6 1936.56  7997.2 1939.58  8056.4 1938.29
  8145.8 1942.20  8196.3 1940.57  8233.9 1943.64  8410.1 1944.70  8651.5 1950.79
#Mann=7,-1,0
  2563.7   0.045       0  4990.7   0.045       0  5028.6   0.045       0
  6750.8   0.035       0  6893.9    0.07       0  7291.4   0.035       0
  7528.9   0.045       0
Bank Sta=4990.7,5028.6
Exp/Cntr=0.3,0.1

Type RM Length L Ch R = 1,24367,634,634,634
BEGIN DESCRIPTION:
Alkali Creek 21.0
END DESCRIPTION:
XS GIS Cut Line= 5
      1383004.41      6969064.13      1382108.86      6966576.49
      1382005.00      6966288.00      1381864.37      6966050.62
      1379805.03      6963888.03
#Sta/Elev= 30
  2049.7 1938.76  2100.9 1937.34  2324.4 1930.96  2772.4 1924.82  3806.7 1924.37
  4233.5 1924.58  4688.5 1925.45  4819.6 1922.93  5003.2 1923.46  5008.1 1923.12
  5010.0 1919.12  5011.0 1918.62  5048.9 1919.12  5050.9 1922.02  5081.6 1923.36
  5217.2 1925.34  5745.4 1923.12  6706.3 1927.05  7335.1 1935.35  7532.7 1936.71
  7576.3 1939.90  7597.7 1938.48  7781.4 1940.57  7816.9 1943.47  7922.9 1942.75
  7979.5 1945.98  8022.0 1944.63  8149.4 1949.29  8198.8 1947.83  8262.4 1950.16
#Mann=11,-1,0
  2049.7    0.07       0  2100.9   0.035       0  2324.4   0.045       0
  3806.7    0.07       0  4233.5   0.045       0  5010.0   0.045       0
  5048.9   0.045       0  5217.2   0.045       0  5745.4    0.07       0
  7335.1   0.035       0  7532.7   0.045       0
Bank Sta=5010,5048.9
Exp/Cntr=0.3,0.1

Type RM Length L Ch R = 1,23733,970,970,970
BEGIN DESCRIPTION:
Alkali Creek 20.5
END DESCRIPTION:
XS GIS Cut Line= 3
      1382898.09      6966567.68      1382528.51      6966065.02
      1382085.28      6965541.70
#Sta/Elev= 30
  4376.1 1941.21  4442.2 1939.72  4456.8 1937.78  4489.0 1937.13  4551.9 1934.41
  4628.1 1933.82  4833.1 1927.27  4861.0 1926.87  4899.7 1924.32  4943.6 1922.79
  4949.9 1921.23  4952.0 1919.02  4953.0 1918.52  4990.9 1919.02  4993.8 1919.90
  5014.5 1919.74  5022.2 1922.21  5028.8 1922.55  5106.6 1922.82  5184.7 1924.28
  5213.3 1927.83  5291.3 1927.59  5319.9 1928.86  5340.7 1931.65  5383.6 1932.44
  5447.3 1936.84  5553.9 1938.35  5631.9 1940.54  5652.7 1942.17  5685.8 1942.36
#Mann=8,-1,0
  4376.1    0.07       0  4489.0   0.035       0  4551.9   0.045       0
  4833.1    0.07       0  4861.0   0.045       0  4952.0   0.045       0
  4990.9   0.045       0  5106.6    0.07       0
Bank Sta=4952,4990.9
Exp/Cntr=0.3,0.1

Type RM Length L Ch R = 1,22763,654,654,654
BEGIN DESCRIPTION:
Alkali Creek 20.0
END DESCRIPTION:
XS GIS Cut Line= 4
      1383052.50      6966673.37      1383194.86      6965639.06
      1383187.05      6965305.73      1384272.97      6963976.76
#Sta/Elev= 30
  3754.8 1942.48  3820.8 1937.77  3946.4 1936.33  4023.6 1933.46  4321.5 1929.40
  4517.3 1929.10  4619.9 1924.68  4638.4 1925.98  4734.3 1923.55  4910.0 1921.14
  4980.0 1923.56  4980.2 1919.12  4981.2 1918.62  5031.0 1919.12  5040.0 1922.80
  5050.0 1923.34  5132.0 1921.01  5264.2 1924.28  5299.3 1927.49  5463.8 1934.17
  6294.4 1934.85  6387.0 1937.52  6508.3 1936.84  6529.1 1939.68  6621.7 1938.47
  6671.3 1942.49  6700.0 1940.76  6735.2 1943.85  6763.9 1942.56  6848.5 1944.95
#Mann=8,-1,0
  3754.8   0.035       0  3946.4    0.07       0  4023.6   0.045       0
  4321.5    0.07       0  4734.3   0.045       0  4980.2   0.045       0
  5031.0   0.045       0  5132.0   0.045       0
Bank Sta=4980.2,5031
Exp/Cntr=0.3,0.1

Type RM Length L Ch R = 1,22109,513,513,513
BEGIN DESCRIPTION:
Alkali Creek 19.0
END DESCRIPTION:
XS GIS Cut Line= 5
      1383064.09      6966679.02      1383623.98      6965722.64
      1383638.09      6965550.11      1383707.79      6965412.48
      1384436.26      6964374.12
#Sta/Elev= 30
  3856.7 1942.48  3903.2 1937.86  3959.7 1937.34  4090.8 1937.88  4150.2 1933.06
  4476.8 1933.67  4530.0 1935.08  4749.7 1929.25  4774.4 1927.08  4861.3 1921.35
  4971.9 1921.34  5016.3 1919.10  5017.3 1918.60  5067.2 1919.10  5070.8 1921.48
  5106.8 1923.49  5130.1 1928.75  5170.9 1928.93  5249.9 1926.02  5279.1 1927.78
  5314.8 1925.60  5329.6 1930.36  5460.1 1930.39  5529.9 1932.74  5832.5 1932.61
  6234.3 1935.97  6326.7 1939.43  6493.2 1939.80  6520.2 1942.36  6560.7 1939.78
#Mann=15,-1,0
  3856.7   0.035       0  3959.7    0.07       0  4150.2   0.045       0
  4476.8    0.07       0  4749.7    0.16       0  4774.4    0.07       0
  4861.3   0.045       0  4971.9    0.07       0  5016.3    0.07       0
  5067.2    0.07       0  5070.8   0.045       0  5106.8    0.07       0
  5170.9   0.045       0  5279.1    0.07       0  5460.1   0.045       0
Bank Sta=5016.3,5067.2
Exp/Cntr=0.3,0.1

Type RM Length L Ch R = 1,21596,543,543,543
BEGIN DESCRIPTION:
Alkali Creek 18.0
END DESCRIPTION:
XS GIS Cut Line= 4
      1383454.99      6966788.01      1383920.57      6966075.79
      1383988.93      6966010.69      1384604.98      6964438.04
#Sta/Elev= 30
  4094.8 1943.03  4289.3 1934.56  4439.9 1933.89  4600.0 1934.30  4751.9 1929.83
  4793.6 1926.33  4870.6 1921.13  4968.4 1920.37  4971.2 1916.55  4972.2 1916.05
  5022.1 1916.55  5025.0 1920.71  5094.6 1920.48  5124.4 1924.81  5130.1 1924.09
  5171.9 1928.66  5208.5 1929.98  5358.6 1932.14  5732.1 1933.88  5835.2 1932.78
  5943.8 1935.38  6003.4 1934.20  6063.3 1937.00  6127.7 1936.17  6190.7 1939.32
  6235.1 1938.12  6491.8 1942.48  6630.1 1942.18  6684.4 1944.25  6729.1 1942.85
#Mann=8,-1,0
  4094.8   0.035       0  4439.9   0.045       0  4793.6    0.07       0
  4870.6   0.045       0  4971.2   0.045       0  5022.1   0.045       0
  5130.1    0.07       0  5358.6   0.045       0
Bank Sta=4971.2,5022.1
Exp/Cntr=0.3,0.1

Type RM Length L Ch R = 1,21053,525,525,525
BEGIN DESCRIPTION:
Alkali Creek 17.0
END DESCRIPTION:
XS GIS Cut Line= 4
      1383555.04      6966837.98      1384288.84      6966396.05
      1384451.60      6966272.35      1384640.20      6964958.65
#Sta/Elev= 30
  4018.8 1942.55  4252.2 1933.48  4444.2 1933.26  4542.1 1934.36  4624.6 1932.43
  4863.5 1919.45  4909.5 1918.46  4999.3 1920.06  5021.3 1917.63  5023.8 1914.93
  5024.8 1914.43  5074.7 1914.93  5078.3 1920.71  5094.3 1922.03  5157.0 1921.62
  5267.1 1925.14  5628.1 1929.92  5710.6 1932.28  5740.9 1931.24  5811.6 1933.22
  5862.1 1932.31  5973.3 1935.23  6003.6 1934.15  6051.4 1936.68  6114.7 1936.24
  6145.0 1939.16  6185.4 1938.18  6256.1 1939.65  6296.5 1942.47  6407.0 1942.23
#Mann=8,-1,0
  4018.8    0.07       0  4444.2   0.035       0  4542.1    0.07       0
  4909.5   0.045       0  5023.8   0.045       0  5074.7   0.045       0
  5157.0    0.07       0  5267.1   0.045       0
Bank Sta=5023.8,5074.7
Exp/Cntr=0.3,0.1

Type RM Length L Ch R = 1,20528,81,81,81
BEGIN DESCRIPTION:
Alkali Creek 16.0
END DESCRIPTION:
XS GIS Cut Line= 4
      1384005.00      6967188.00      1384645.14      6966980.26
      1384884.72      6965886.51      1384702.90      6965006.69
#Sta/Elev= 30
  3875.6 1942.10  4056.7 1932.32  4262.2 1925.63  4581.6 1921.64  4754.4 1921.59
  4960.4 1919.21  4980.9 1918.02  4986.1 1914.32  4987.1 1913.82  5037.0 1914.32
  5037.9 1917.50  5043.0 1918.73  5093.5 1920.94  5599.8 1925.96  5758.7 1928.66
  5776.9 1930.80  5860.8 1930.37  5962.9 1933.14  5993.5 1931.96  6054.8 1932.70
  6146.7 1935.51  6189.2 1934.30  6239.4 1936.94  6310.1 1936.36  6350.9 1939.47
  6385.0 1938.27  6442.8 1939.58  6480.4 1942.71  6504.1 1941.47  6566.7 1942.10
#Mann=5,-1,0
  3875.6    0.07       0  4262.2   0.035       0  4986.1   0.035       0
  5037.0   0.035       0  5776.9   0.045       0
Bank Sta=4986.1,5037
Exp/Cntr=0.3,0.1

Type RM Length L Ch R = 1,20447,532,532,532
BEGIN DESCRIPTION:
Alkali Creek 15.5
END DESCRIPTION:
XS GIS Cut Line= 4
      1384182.04      6967492.28      1384705.90      6967079.22
      1384937.13      6965957.09      1384900.67      6965084.68
#Sta/Elev= 30
  3827.5 1941.87  3882.2 1941.27  4010.0 1931.40  4018.0 1932.35  4024.4 1929.78
  4032.5 1931.00  4046.9 1928.88  4252.1 1923.29  4926.6 1918.63  4954.3 1918.64
  4996.2 1919.09  5010.9 1917.34  5011.6 1913.71  5012.6 1913.21  5062.5 1913.71
  5067.6 1920.17  5231.0 1920.12  5282.0 1922.91  5357.9 1922.45  5373.9 1924.97
  5403.1 1923.27  5476.0 1923.68  5516.9 1926.35  5619.0 1925.06  5769.5 1929.00
  5807.9 1928.26  5829.6 1930.89  6098.1 1932.74  6440.1 1936.64  6513.5 1939.16
#Mann=6,-1,0
  3827.5   0.035       0  4926.6    0.07       0  4954.3   0.035       0
  5011.6   0.035       0  5062.5   0.035       0  6098.1   0.045       0
Bank Sta=5011.6,5062.5
Exp/Cntr=0.3,0.1

Type RM Length L Ch R = 1,19915,528,528,528
BEGIN DESCRIPTION:
Alkali Creek 15.0
END DESCRIPTION:
XS GIS Cut Line= 4
      1384254.07      6967597.77      1385254.47      6966806.90
      1385317.40      6966716.50      1385469.11      6965771.80
#Sta/Elev= 30
  3674.8 1942.58  3685.4 1942.46  3708.6 1940.95  3917.7 1929.09  4045.7 1924.01
  4173.1 1923.69  4232.6 1921.12  4799.6 1917.81  4972.1 1919.09  4985.3 1917.85
  4988.5 1912.30  4989.5 1911.80  5039.5 1912.30  5043.7 1918.64  5084.3 1918.80
  5218.9 1922.43  5266.0 1923.97  5311.9 1922.08  5518.8 1922.48  5544.8 1925.36
  5595.5 1922.74  5656.2 1926.63  5686.6 1924.22  5808.2 1924.92  5848.7 1927.89
  5900.4 1926.12  5929.7 1928.86  5962.3 1927.61  5990.5 1930.70  6017.0 1929.33
#Mann=10,-1,0
  3674.8    0.07       0  3685.4   0.035       0  3708.6    0.07       0
  3917.7   0.035       0  4232.6   0.045       0  4799.6    0.07       0
  4988.5    0.07       0  5039.5    0.07       0  5084.3    0.16       0
  5218.9   0.045       0
Bank Sta=4988.5,5039.5
Exp/Cntr=0.3,0.1

Type RM Length L Ch R = 1,19387,501,501,501
BEGIN DESCRIPTION:
Alkali Creek 14.0
END DESCRIPTION:
XS GIS Cut Line= 4
      1384482.32      6968089.78      1384977.13      6967268.58
      1385365.58      6967068.06      1386058.75      6967284.22
#Sta/Elev= 30
  3562.4 1950.86  3707.7 1942.48  3901.2 1932.40  4119.4 1924.53  4298.2 1921.04
  4336.9 1920.25  4368.0 1921.51  4404.9 1919.50  4518.8 1918.67  4743.8 1917.33
  4839.0 1918.02  4855.5 1917.67  4867.6 1916.26  4890.1 1918.10  4922.0 1917.07
  4968.2 1918.08  4979.4 1917.18  4986.4 1911.82  4987.4 1911.32  5037.4 1911.82
  5039.2 1917.56  5044.4 1918.71  5087.4 1918.76  5244.7 1918.68  5370.3 1922.74
  5469.2 1927.80  5477.5 1929.00  5523.3 1930.37  5586.2 1934.83  5684.4 1944.94
#Mann=10,-1,0
  3562.4   0.035       0  3707.7    0.07       0  3901.2   0.045       0
  4298.2    0.07       0  4518.8   0.045       0  4986.4   0.045       0
  5037.4   0.045       0  5087.4    0.07       0  5370.3    0.16       0
  5469.2    0.07       0
Bank Sta=4986.4,5037.4
Exp/Cntr=0.3,0.1

Type RM Length L Ch R = 1,18886,526,526,526
BEGIN DESCRIPTION:
Alkali Creek 13.0
END DESCRIPTION:
XS GIS Cut Line= 5
      1384954.97      6967938.04      1385283.87      6967526.91
      1385355.00      6967438.00      1385430.00      6967363.00
      1386041.29      6967344.29
#Sta/Elev= 30
  4359.9 1937.78  4509.6 1930.00  4565.6 1928.08  4602.5 1925.22  4768.3 1920.74
  4852.1 1919.44  4890.9 1917.86  4964.2 1917.43  4967.6 1911.65  4968.6 1911.15
  5018.6 1911.65  5028.5 1917.81  5042.7 1917.11  5121.3 1918.14  5142.4 1917.57
  5151.3 1917.56  5171.4 1913.98  5181.4 1914.45  5191.4 1917.06  5241.6 1917.83
  5301.4 1918.71  5340.7 1921.31  5490.0 1928.75  5502.6 1929.24  5521.5 1929.60
  5571.5 1933.14  5581.5 1935.15  5621.6 1937.59  5711.6 1945.37  5717.9 1944.17
#Mann=11,-1,0
  4359.9   0.045       0  4768.3   0.035       0  4852.1    0.07       0
  4890.9   0.035       0  4967.6   0.035       0  5018.6    0.07       0
  5142.4   0.045       0  5241.6    0.16       0  5340.7    0.07       0
  5490.0    0.16       0  5502.6    0.07       0
Bank Sta=4967.6,5018.6
Exp/Cntr=0.3,0.1

Type RM Length L Ch R = 1,18360,532,532,532
BEGIN DESCRIPTION:
Alkali Creek 12.0
END DESCRIPTION:
XS GIS Cut Line= 3
      1384502.74      6968138.30      1385765.23      6967729.58
      1386000.36      6967403.52
#Sta/Elev= 30
  3736.1 1950.81  3767.9 1949.95  3883.9 1943.79  3893.8 1943.42  3981.2 1940.13
  4308.3 1936.64  4652.9 1920.83  4716.0 1920.21  4831.6 1916.28  4924.7 1916.15
  4958.8 1916.37  4964.8 1911.74  4965.8 1911.24  5016.8 1911.74  5017.5 1915.91
  5049.5 1919.57  5054.8 1918.79  5060.4 1920.75  5071.2 1920.27  5092.1 1921.95
  5100.7 1918.01  5106.8 1922.17  5121.5 1922.32  5127.7 1925.18  5151.0 1928.85
  5207.4 1934.30  5293.3 1939.22  5328.9 1939.38  5373.1 1942.17  5465.1 1944.94
#Mann=8,-1,0
  3736.1   0.035       0  3767.9    0.07       0  3883.9   0.045       0
  3893.8    0.07       0  3981.2   0.045       0  4924.7    0.07       0
  4964.8    0.07       0  5016.8    0.07       0
Bank Sta=4964.8,5016.8
Exp/Cntr=0.3,0.1

Type RM Length L Ch R = 1,17828,406,406,406
BEGIN DESCRIPTION:
Alkali Creek 11.0
END DESCRIPTION:
XS GIS Cut Line= 4
      1384762.35      6968353.09      1385698.62      6968278.04
      1385903.78      6968159.13      1386005.00      6967438.00
#Sta/Elev= 30
  3937.7 1936.07  4000.6 1933.47  4482.5 1928.59  4662.7 1927.54  4712.8 1924.22
  4763.0 1923.53  4823.2 1920.33  4882.8 1919.95  4921.9 1917.55  4976.8 1915.13
  4984.7 1916.23  4986.0 1910.74  4987.0 1910.24  5038.0 1910.74  5038.3 1911.05
  5043.5 1916.42  5049.3 1916.71  5145.8 1915.41  5244.2 1916.72  5426.5 1920.01
  5441.1 1920.56  5539.4 1923.67  5650.4 1929.99  5664.0 1929.57  5690.8 1932.85
  5771.6 1937.34  5791.8 1940.34  5801.6 1941.04  5806.6 1939.22  5842.3 1942.33
#Mann=10,-1,0
  3937.7   0.045       0  4482.5    0.07       0  4921.9    0.16       0
  4986.0   0.045       0  5038.0    0.16       0  5038.3    0.16       0
  5145.8   0.045       0  5244.2    0.07       0  5426.5   0.045       0
  5441.1    0.07       0
Bank Sta=4986,5038
Exp/Cntr=0.3,0.1

Type RM Length L Ch R = 1,17422,729,729,729
BEGIN DESCRIPTION:
Alkali Creek 10.3
END DESCRIPTION:
XS GIS Cut Line= 4
      1385668.63      6969058.79      1386181.55      6968449.93
      1386126.00      6968238.13      1386087.80      6967345.73
#Sta/Elev= 30
  4088.6 1926.92  4214.4 1927.68  4263.8 1925.17  4327.5 1925.55  4356.1 1923.72
  4448.5 1921.05  4491.4 1921.88  4561.6 1919.12  4647.5 1919.00  4690.3 1919.89
  4711.1 1918.58  4837.5 1917.33  4972.1 1915.30  4974.4 1910.35  4975.4 1909.85
  5026.4 1910.35  5031.5 1915.94  5110.2 1914.91  5208.2 1915.85  5306.3 1916.82
  5502.5 1919.49  5574.2 1921.36  5644.3 1924.89  5654.3 1926.43  5693.3 1927.25
  5781.0 1932.18  5864.5 1936.29  5904.5 1939.58  5942.5 1940.35  5996.9 1944.17
#Mann=11,-1,0
  4088.6   0.045       0  4647.5    0.07       0  4837.5    0.16       0
  4974.4    0.07       0  5026.4    0.16       0  5110.2    0.16       0
  5208.2    0.07       0  5306.3   0.045       0  5502.5    0.07       0
  5693.3   0.045       0  5781.0    0.07       0
Bank Sta=4974.4,5026.4
Exp/Cntr=0.3,0.1

Type RM Length L Ch R = 1,16693,330,330,330
BEGIN DESCRIPTION:
Alkali Creek 10.25
END DESCRIPTION:
XS GIS Cut Line= 4
      1386830.01      6968863.04      1386565.56      6968080.15
      1386467.57      6967671.18      1386130.00      6967213.00
#Sta/Elev= 30
  3872.7 1925.48  3930.3 1926.05  3973.0 1925.48  4036.3 1920.59  4187.3 1917.52
  4321.3 1917.94  4395.2 1916.79  4416.3 1917.79  4448.0 1916.40  4511.3 1916.15
  4685.9 1916.87  4783.5 1914.80  4982.2 1914.76  4989.2 1913.74  4991.4 1912.06
  4993.1 1910.76  4994.1 1910.26  5045.1 1910.76  5050.9 1916.99  5061.1 1917.16
  5071.5 1921.26  5092.0 1925.25  5187.4 1931.47  5226.4 1931.49  5417.2 1933.75
  5496.2 1936.07  5562.4 1939.87  5582.2 1940.30  5638.6 1944.86  5688.7 1945.49
#Mann=8,-1,0
  3872.7   0.045       0  3930.3    0.07       0  4685.9   0.045       0
  4991.4    0.07       0  4993.1    0.07       0  5045.1    0.07       0
  5226.4   0.045       0  5562.4    0.07       0
Bank Sta=4993.1,5045.1
Exp/Cntr=0.3,0.1

Type RM Length L Ch R = 1,16363,715,715,715
BEGIN DESCRIPTION:
Alkali Creek 10.2
END DESCRIPTION:
XS GIS Cut Line= 5
      1387263.61      6968601.88      1386805.25      6967917.82
      1386815.67      6967706.01      1386749.70      6967230.32
      1386850.20      6966814.43
#Sta/Elev= 30
  4093.9 1931.17  4138.5 1930.03  4231.6 1923.84  4282.6 1921.40  4355.5 1919.52
  4411.7 1917.86  4669.4 1915.08  4744.8 1914.77  4759.8 1915.06  4765.9 1916.16
  4786.9 1915.49  4831.9 1915.97  4844.0 1915.19  4977.2 1914.33  4987.1 1910.25
  4988.1 1909.75  5039.1 1910.25  5047.3 1914.25  5113.0 1914.90  5202.4 1916.29
  5258.6 1917.17  5440.4 1917.02  5734.5 1919.19  5739.6 1919.95  5756.1 1919.67
  5781.5 1920.82  5823.4 1920.75  5941.2 1923.06  5990.8 1925.81  6037.5 1925.70
#Mann=8,-1,0
  4093.9    0.07       0  4355.5   0.045       0  4669.4    0.07       0
  4844.0   0.045       0  4987.1   0.045       0  5039.1   0.045       0
  5113.0    0.07       0  5202.4   0.045       0
Bank Sta=4987.1,5039.1
Exp/Cntr=0.3,0.1

Type RM Length L Ch R = 1,15648,625,625,625
BEGIN DESCRIPTION:
Alkali Creek 10.1
END DESCRIPTION:
XS GIS Cut Line= 3
      1387628.16      6968086.98      1387428.28      6967700.19
      1387135.99      6967004.48
#Sta/Elev= 30
  4333.6 1932.44  4394.6 1931.65  4433.3 1930.36  4438.9 1929.52  4483.2 1928.51
  4499.8 1928.72  4505.4 1927.96  4535.1 1927.06  4588.3 1926.18  4638.3 1923.62
  4670.1 1923.30  4726.9 1920.27  4772.9 1919.66  4819.9 1917.38  4879.1 1914.93
  4938.1 1914.16  4947.8 1914.53  4966.1 1912.66  4969.2 1910.23  4970.3 1909.73
  5020.4 1909.73  5021.4 1910.23  5024.5 1913.64  5064.2 1915.05  5140.1 1915.51
  5225.4 1919.75  5292.0 1924.28  5389.6 1929.77  5443.8 1931.68  5523.6 1932.29
#Mann=6,-1,0
  4333.6    0.07       0  4819.9   0.045       0  4879.1    0.07       0
  4938.1   0.045       0  4969.2   0.045       0  5021.4   0.045       0
Bank Sta=4969.2,5021.4
Exp/Cntr=0.3,0.1

Type RM Length L Ch R = 1,15023,788,788,788
BEGIN DESCRIPTION:
Alkali Creek 10.0
END DESCRIPTION:
XS GIS Cut Line= 4
      1387677.74      6968068.41      1387830.08      6967570.16
      1387805.00      6967433.01      1388070.25      6966645.63
#Sta/Elev= 30
  4396.9 1933.18  4507.2 1933.15  4585.9 1931.66  4839.3 1917.52  4867.9 1916.02
  4921.8 1915.22  4940.4 1913.74  4948.9 1910.58  4949.9 1910.08  5001.1 1910.58
  5193.9 1918.70  5221.5 1919.98  5264.7 1921.38  5347.5 1928.53  5390.6 1928.69
  5416.8 1931.75  5442.5 1931.60  5448.3 1932.66  5453.6 1931.95  5474.2 1934.69
  5495.3 1934.65  5511.3 1936.43  5548.1 1936.50  5569.0 1938.92  5621.9 1939.10
  5653.6 1941.55  5716.9 1941.20  5763.2 1942.23  5789.4 1943.88  5888.2 1944.18
#Mann=7,-1,0
  4396.9    0.07       0  4585.9   0.045       0  4839.3    0.07       0
  4948.9   0.045       0  5001.1    0.07       0  5193.9    0.07       0
  5221.5   0.045       0
Bank Sta=4948.9,5001.1
Exp/Cntr=0.3,0.1

Type RM Length L Ch R = 1,14235,712,712,712
BEGIN DESCRIPTION:
Alkali Creek 9.8
END DESCRIPTION:
XS GIS Cut Line= 3
      1387653.41      6968216.87      1387874.89      6968042.95
      1388969.12      6967628.47
#Sta/Elev= 30
  4264.8 1932.87  4278.4 1932.86  4485.4 1931.92  4528.8 1929.64  4579.2 1928.65
  4701.3 1923.03  4706.2 1922.89  4820.1 1916.55  4845.9 1915.83  4854.0 1916.69
  4884.2 1912.28  4909.0 1911.14  4939.2 1913.20  4944.5 1912.41  4948.6 1908.19
  4949.6 1907.69  5000.8 1908.19  5006.3 1912.06  5017.0 1912.30  5026.1 1911.43
  5054.4 1912.31  5059.8 1913.66  5114.7 1913.25  5146.3 1915.49  5273.7 1918.99
  5348.5 1923.34  5389.6 1923.52  5425.1 1926.08  5510.0 1926.33  5716.5 1926.26
#Mann=10,-1,0
  4264.8    0.07       0  4278.4   0.045       0  4701.3    0.07       0
  4706.2   0.045       0  4820.1    0.07       0  4948.6    0.07       0
  5000.8    0.07       0  5026.1   0.045       0  5146.3    0.07       0
  5510.0   0.045       0
Bank Sta=4948.6,5000.8
Exp/Cntr=0.3,0.1

Type RM Length L Ch R = 1,13523,531,531,531
BEGIN DESCRIPTION:
Alkali Creek 9.7
END DESCRIPTION:
XS GIS Cut Line= 4
      1387762.58      6968400.84      1388052.65      6968472.51
      1388606.96      6968590.55      1388790.20      6968505.61
#Sta/Elev= 30
  4432.2 1932.68  4506.8 1931.52  4582.1 1927.78  4694.4 1922.51  4780.4 1917.37
  4835.6 1916.31  4845.9 1915.60  4866.3 1912.86  4879.5 1912.11  4886.8 1912.49
  4907.2 1911.21  4929.1 1911.13  4937.9 1911.73  4948.1 1911.25  4958.3 1912.19
  4978.8 1910.94  4980.6 1909.34  4983.3 1906.93  4984.3 1906.43  5034.5 1906.43
  5035.5 1906.93  5040.1 1910.21  5045.0 1910.49  5060.6 1912.20  5111.7 1912.13
  5190.0 1915.27  5260.7 1918.94  5350.7 1921.76  5382.6 1923.43  5499.7 1923.34
#Mann=7,-1,0
  4432.2   0.045       0  4582.1    0.07       0  4980.6    0.16       0
  4983.3    0.07       0  5035.5    0.16       0  5045.0    0.07       0
  5190.0   0.045       0
Bank Sta=4983.3,5035.5
Exp/Cntr=0.3,0.1

Type RM Length L Ch R = 1,12992,742,742,742
BEGIN DESCRIPTION:
Alkali Creek 9.6
END DESCRIPTION:
XS GIS Cut Line= 4
      1387548.28      6968362.00      1387930.34      6968952.97
      1388330.92      6969054.09      1389139.64      6968890.32
#Sta/Elev= 30
  4064.4 1932.47  4071.2 1932.50  4196.5 1931.98  4232.8 1930.78  4428.8 1928.85
  4597.7 1923.37  4635.9 1922.73  4725.6 1919.72  4761.9 1917.56  4824.5 1916.53
  4833.0 1915.37  4834.4 1915.18  4850.1 1913.27  4896.7 1911.83  4932.2 1911.40
  4958.6 1912.78  4973.3 1911.78  4973.7 1905.49  4974.7 1904.99  5025.9 1905.49
  5030.8 1911.31  5061.7 1910.55  5113.3 1911.36  5202.9 1914.30  5239.3 1915.06
  5348.7 1920.15  5430.3 1921.98  5532.3 1920.47  5634.4 1920.43  6006.4 1921.85
#Mann=9,-1,0
  4064.4    0.07       0  4071.2   0.045       0  4597.7    0.07       0
  4635.9   0.045       0  4833.0    0.07       0  4834.4    0.16       0
  4973.7    0.07       0  5025.9    0.16       0  5202.9   0.045       0
Bank Sta=4973.7,5025.9
Exp/Cntr=0.3,0.1

Type RM Length L Ch R = 1,12250,690,690,690
BEGIN DESCRIPTION:
Alkali Creek 9.5
END DESCRIPTION:
XS GIS Cut Line= 4
      1387529.98      6969863.02      1387758.83      6969684.36
      1388144.62      6969649.31      1388836.12      6969289.55
#Sta/Elev= 30
  4512.7 1923.50  4620.3 1922.35  4697.3 1919.67  4755.1 1919.81  4797.4 1918.01
  4843.1 1917.41  4859.4 1917.44  4879.5 1918.62  4909.6 1915.88  4942.7 1914.91
  4959.8 1913.52  4979.9 1910.91  4983.9 1905.51  4984.9 1905.01  5035.1 1905.01
  5036.2 1905.51  5037.1 1909.24  5042.2 1908.92  5050.2 1910.78  5100.4 1910.28
  5110.8 1910.87  5140.6 1910.21  5193.4 1910.64  5223.3 1911.89  5281.0 1913.74
  5310.8 1915.88  5316.4 1915.47  5374.5 1916.57  5554.0 1919.77  5969.9 1919.81
#Mann=8,-1,0
  4512.7   0.045       0  4843.1    0.07       0  4942.7    0.16       0
  4983.9    0.07       0  5036.2    0.16       0  5110.8    0.16       0
  5223.3    0.07       0  5374.5   0.045       0
Bank Sta=4983.9,5036.2
Exp/Cntr=0.3,0.1

Type RM Length L Ch R = 1,11560,679,679,679
BEGIN DESCRIPTION:
Alkali Creek 9.4
END DESCRIPTION:
XS GIS Cut Line= 3
      1387430.01      6971112.99      1388248.25      6970231.54
      1388836.53      6969435.65
#Sta/Elev= 30
  3797.3 1920.73  3889.1 1920.68  3945.8 1919.19  4016.7 1919.29  4073.4 1918.10
  4271.2 1917.83  4370.4 1919.03  4554.6 1918.65  4775.5 1915.05  4801.9 1916.12
  4823.4 1913.93  4865.9 1912.17  4936.6 1911.08  4938.4 1906.34  4939.5 1905.84
  4990.7 1906.34  4992.9 1909.37  5021.4 1908.42  5029.3 1910.35  5050.7 1910.88
  5065.3 1910.15  5071.5 1910.80  5079.0 1910.03  5165.5 1909.68  5278.2 1912.27
  5286.6 1913.22  5307.4 1912.55  5391.7 1915.14  5700.8 1919.62  5989.7 1919.91
#Mann=5,-1,0
  3797.3   0.045       0  4775.5    0.07       0  4938.4    0.07       0
  4990.7    0.07       0  5391.7   0.045       0
Bank Sta=4938.4,4990.7
Exp/Cntr=0.3,0.1

Type RM Length L Ch R = 1,10881,304,304,304
BEGIN DESCRIPTION:
Alkali Creek 9.3
END DESCRIPTION:
XS GIS Cut Line= 3
      1388233.30      6970981.60      1388868.71      6970275.02
      1388927.56      6969611.39
#Sta/Elev= 30
  4174.8 1919.15  4285.0 1917.14  4327.6 1917.12  4454.7 1914.53  4617.6 1913.07
  4627.8 1913.63  4635.0 1913.47  4688.6 1912.80  4723.8 1911.53  4766.4 1911.33
  4773.1 1910.62  4801.5 1910.82  4808.9 1909.73  4944.9 1909.70  4978.6 1909.92
  4986.1 1908.69  4987.6 1903.62  4988.6 1903.12  5038.9 1903.12  5039.9 1903.62
  5042.2 1908.54  5063.9 1910.26  5125.1 1911.48  5143.4 1912.97  5222.5 1914.45
  5255.3 1916.02  5292.7 1915.09  5350.7 1916.31  5624.0 1920.64  5791.3 1920.69
#Mann=8,-1,0
  4174.8   0.045       0  4627.8    0.07       0  4635.0   0.045       0
  4808.9    0.16       0  4944.9    0.07       0  4987.6    0.07       0
  5039.9    0.07       0  5350.7   0.045       0
Bank Sta=4987.6,5039.9
Exp/Cntr=0.3,0.1

Type RM Length L Ch R = 1,10577,111,111,111
BEGIN DESCRIPTION:
Alkali Creek 9.25
END DESCRIPTION:
XS GIS Cut Line= 2
      1388842.95      6971612.45      1389240.81      6969016.96
#Sta/Elev= 30
  3959.2 1921.84  4070.8 1922.19  4075.9 1920.25  4134.2 1921.73  4139.2 1919.55
  4202.6 1920.97  4207.6 1919.03  4265.9 1920.54  4271.0 1918.67  4327.9 1919.60
  4339.4 1917.32  4597.9 1913.48  4798.0 1913.02  4861.4 1910.41  4866.4 1911.74
  4904.6 1908.38  4985.5 1907.21  4989.6 1903.82  4990.7 1903.32  5042.0 1903.82
  5046.2 1908.07  5061.5 1908.69  5066.6 1911.10  5117.0 1910.04  5129.9 1911.81
  5238.4 1911.80  5380.1 1915.53  5525.2 1916.08  5774.6 1921.70  6585.0 1921.47
#Mann=3,-1,0
  3959.2   0.035       0  4989.6   0.035       0  5042.0   0.035       0
Bank Sta=4989.6,5042
Exp/Cntr=0.3,0.1

Type RM Length L Ch R = 1,10466,316,316,316
BEGIN DESCRIPTION:
Alkali Creek 9.22
END DESCRIPTION:
XS GIS Cut Line= 2
      1388915.86      6971638.54      1389346.60      6969052.36
#Sta/Elev= 30
  4009.6 1920.89  4582.8 1913.69  4760.2 1914.03  4765.3 1911.77  4821.1 1912.84
  4826.2 1910.74  4881.9 1912.53  4887.0 1910.02  4942.8 1911.84  4947.8 1908.80
  4993.5 1907.17  4997.7 1903.40  4998.8 1902.90  5050.1 1903.40  5054.3 1908.61
  5130.4 1913.43  5135.5 1911.87  5191.2 1913.40  5196.3 1911.94  5252.1 1913.21
  5257.2 1911.67  5378.8 1912.71  5617.2 1917.04  5622.2 1918.41  5678.0 1917.63
  5738.9 1918.70  5743.9 1920.07  5916.0 1920.93  5926.5 1922.27  6631.4 1920.87
#Mann=3,-1,0
  4009.6   0.035       0  4997.7   0.035       0  5050.1   0.035       0
Bank Sta=4997.7,5050.1
Exp/Cntr=0.3,0.1

Type RM Length L Ch R = 1,10150,553,553,553
BEGIN DESCRIPTION:
Alkali Creek 9.2
END DESCRIPTION:
XS GIS Cut Line= 3
      1389549.46      6971257.53      1389287.76      6970649.76
      1389389.48      6969064.54
#Sta/Elev= 30
  4419.0 1929.50  4496.8 1929.68  4549.3 1925.94  4590.9 1926.21  4608.4 1924.49
  4625.4 1922.84  4667.0 1922.73  4701.6 1919.48  4734.2 1919.32  4772.0 1916.12
  4819.0 1915.53  4877.0 1910.19  4918.6 1911.03  4952.8 1907.03  4973.4 1906.82
  4984.7 1906.98  4991.1 1902.63  4992.1 1902.13  5043.5 1902.63  5047.2 1908.16
  5323.0 1910.79  5421.7 1910.28  5483.3 1909.68  5586.3 1911.63  5739.6 1917.62
  5914.2 1921.77  6051.1 1922.78  6335.1 1919.77  6596.2 1920.09  6669.2 1920.89
#Mann=8,-1,0
  4419.0   0.035       0  4608.4    0.07       0  4952.8    0.16       0
  4973.4    0.07       0  4991.1    0.07       0  5043.5    0.07       0
  5421.7   0.045       0  6596.2   0.035       0
Bank Sta=4991.1,5043.5
Exp/Cntr=0.3,0.1

Type RM Length L Ch R = 1,9597,648,648,648
BEGIN DESCRIPTION:
Alkali Creek 9.1
END DESCRIPTION:
XS GIS Cut Line= 3
      1389557.29      6971182.04      1389731.83      6970546.51
      1389406.84      6968856.13
#Sta/Elev= 30
  4176.9 1929.55  4340.0 1926.23  4394.7 1922.87  4471.5 1922.57  4533.7 1919.16
  4567.4 1920.07  4601.8 1916.79  4658.1 1914.92  4720.7 1915.18  4782.6 1912.64
  4829.1 1913.42  4847.7 1911.15  4899.4 1909.76  4966.8 1907.96  4977.0 1906.69
  4982.4 1900.88  4983.4 1900.38  5034.8 1900.88  5038.1 1904.65  5068.7 1908.74
  5139.9 1907.39  5290.7 1909.27  5400.4 1912.11  5476.0 1915.80  5496.4 1918.88
  5542.3 1919.42  5659.3 1921.22  5720.4 1919.75  6493.5 1920.62  6557.3 1921.62
#Mann=9,-1,0
  4176.9   0.035       0  4394.7    0.07       0  4899.4    0.16       0
  4982.4    0.07       0  5034.8    0.16       0  5290.7   0.045       0
  5400.4    0.07       0  5542.3   0.045       0  6493.5   0.035       0
Bank Sta=4982.4,5034.8
Exp/Cntr=0.3,0.1

Type RM Length L Ch R = 1,8949,413,413,413
BEGIN DESCRIPTION:
Alkali Creek 9.0
END DESCRIPTION:
XS GIS Cut Line= 5
      1389578.40      6971204.77      1390136.78      6970222.10
      1390155.00      6970138.00      1390166.29      6970020.71
      1389559.57      6968865.57
#Sta/Elev= 30
  3783.3 1930.21  3888.3 1929.70  3947.1 1926.08  3984.9 1926.67  4028.2 1923.61
  4114.6 1922.63  4159.1 1919.78  4431.8 1916.40  4584.7 1908.98  4620.7 1910.42
  4714.5 1907.94  4958.7 1906.47  4963.2 1900.35  4964.2 1899.85  5015.6 1900.35
  5019.7 1906.67  5024.7 1906.62  5116.3 1910.53  5150.6 1908.55  5299.3 1909.65
  5343.4 1912.17  5365.4 1910.94  5409.5 1913.38  5448.0 1912.72  5475.7 1915.06
  5514.1 1914.23  5549.7 1916.69  5607.9 1915.67  5690.5 1918.11  6422.2 1920.40
#Mann=6,-1,0
  3783.3   0.035       0  3947.1    0.07       0  4714.5    0.16       0
  4963.2    0.07       0  5015.6    0.16       0  5024.7   0.045       0
Bank Sta=4963.2,5015.6
Exp/Cntr=0.3,0.1

Type RM Length L Ch R = 1,8536,538,538,538
BEGIN DESCRIPTION:
Alkali Creek 8.5
END DESCRIPTION:
XS GIS Cut Line= 3
      1389619.78      6971192.48      1390656.25      6970145.59
      1390406.87      6969571.49
#Sta/Elev= 30
  3734.8 1930.32  3828.8 1928.99  3861.9 1926.23  3911.3 1926.43  4088.2 1919.66
  4314.4 1915.79  4342.7 1916.92  4413.4 1913.68  4448.8 1914.78  4477.0 1912.23
  4611.4 1910.15  4646.8 1907.18  4752.9 1908.41  4795.3 1906.15  4874.8 1906.16
  4972.0 1905.97  4979.1 1904.71  4981.2 1898.02  4982.2 1897.52  5033.7 1898.02
  5035.7 1905.09  5042.8 1905.84  5137.1 1906.30  5241.0 1906.39  5368.8 1910.43
  5403.2 1909.42  5450.1 1912.17  5578.3 1912.89  5630.6 1915.58  5833.9 1916.48
#Mann=7,-1,0
  3734.8   0.035       0  3828.8    0.07       0  4874.8   0.045       0
  4981.2   0.045       0  5033.7   0.045       0  5137.1    0.07       0
  5241.0   0.045       0
Bank Sta=4981.2,5033.7
Exp/Cntr=0.3,0.1

Type RM Length L Ch R = 1,7998,503,503,503
BEGIN DESCRIPTION:
Alkali Creek 8.4
END DESCRIPTION:
XS GIS Cut Line= 4
      1389640.59      6971192.48      1390983.61      6970529.93
      1391035.82      6970134.62      1390680.02      6969513.04
#Sta/Elev= 30
  3258.4 1930.71  3326.1 1929.72  3487.6 1922.87  3549.4 1922.88  3706.5 1917.46
  3841.2 1916.71  3863.7 1914.76  3981.5 1914.84  4055.0 1911.76  4088.2 1912.76
  4295.9 1907.90  4458.6 1908.31  4655.1 1903.70  4776.6 1905.84  4939.5 1905.57
  4969.7 1903.65  4973.7 1897.39  4974.8 1896.89  5026.2 1897.39  5029.5 1905.00
  5060.5 1906.39  5173.8 1904.80  5328.4 1907.45  5358.2 1906.08  5548.6 1912.08
  5586.0 1911.03  5634.9 1913.82  5666.6 1912.69  5752.9 1915.56  5870.9 1915.23
#Mann=5,-1,0
  3258.4   0.035       0  3326.1    0.07       0  4776.6   0.045       0
  4973.7   0.045       0  5026.2   0.045       0
Bank Sta=4973.7,5026.2
Exp/Cntr=0.3,0.1

Type RM Length L Ch R = 1,7495,697,697,697
BEGIN DESCRIPTION:
Alkali Creek 8.3
END DESCRIPTION:
XS GIS Cut Line= 4
      1389658.89      6971200.26      1391464.42      6970488.48
      1391498.21      6970178.77      1391114.78      6969166.89
#Sta/Elev= 30
  2857.2 1930.46  2910.9 1929.47  2986.7 1926.17  3035.5 1926.30  3089.5 1922.73
  3272.2 1919.52  3304.5 1917.08  3573.2 1914.46  3648.4 1911.80  3671.5 1913.08
  3755.9 1909.64  3798.8 1910.59  3828.6 1908.40  3927.9 1908.27  3960.2 1906.34
  4260.5 1904.52  4476.1 1903.89  4508.0 1905.47  4562.1 1903.76  4943.0 1903.18
  4949.3 1903.05  4953.3 1898.24  4954.3 1897.74  5005.8 1898.24  5009.7 1903.59
  5665.0 1905.28  5920.3 1910.02  6030.0 1909.84  6083.5 1912.30  6191.6 1911.45
#Mann=5,-1,0
  2857.2   0.035       0  2910.9    0.07       0  4260.5   0.045       0
  4953.3   0.045       0  5005.8   0.045       0
Bank Sta=4953.3,5005.8
Exp/Cntr=0.3,0.1

Type RM Length L Ch R = 1,6798,293,293,293
BEGIN DESCRIPTION:
Alkali Creek 8.2
END DESCRIPTION:
XS GIS Cut Line= 4
      1389681.82      6971210.27      1391648.44      6970622.16
      1392067.60      6970650.84      1393529.96      6970163.01
#Sta/Elev= 30
  2639.5 1930.14  2676.2 1929.57  2862.0 1923.25  2935.1 1922.81  2987.3 1919.55
  3046.7 1919.65  3112.5 1916.40  3175.1 1916.79  3300.4 1913.50  3332.5 1914.67
  3404.8 1911.65  3437.0 1912.94  3464.9 1910.68  3561.3 1910.41  3613.5 1907.55
  3976.1 1904.10  4135.7 1903.57  4177.1 1905.43  4235.0 1903.26  4889.2 1903.27
  4979.4 1902.05  4983.2 1897.56  4984.3 1897.06  5035.7 1897.56  5039.5 1900.93
  5049.6 1902.28  5089.7 1903.51  6585.4 1905.13  6627.6 1905.70  6653.9 1910.61
#Mann=5,-1,0
  2639.5   0.035       0  2676.2    0.07       0  3976.1   0.045       0
  4983.2   0.045       0  5035.7   0.045       0
Bank Sta=4983.2,5035.7
Exp/Cntr=0.3,0.1

Type RM Length L Ch R = 1,6505,337,337,337
BEGIN DESCRIPTION:
Alkali Creek 8.1
END DESCRIPTION:
XS GIS Cut Line= 4
      1389706.99      6971217.98      1391655.09      6970778.63
      1391930.00      6970918.19      1393421.52      6970629.18
#Sta/Elev= 30
  2884.7 1929.73  2901.2 1929.48  2944.2 1929.61  2999.4 1926.24  3056.9 1926.31
  3097.9 1923.60  3354.2 1916.41  3559.2 1914.38  3635.4 1911.41  3661.7 1912.78
  3692.5 1910.42  3784.8 1910.26  3861.8 1907.17  3897.5 1908.25  3953.3 1905.77
  4135.9 1904.32  4307.6 1903.42  4338.3 1905.25  4379.3 1902.88  4961.7 1902.47
  4967.5 1896.98  4968.6 1896.48  5020.0 1896.98  5022.9 1900.33  5028.5 1902.05
  5095.3 1902.79  5755.4 1901.98  6590.6 1904.29  6682.3 1905.27  6709.3 1909.90
#Mann=5,-1,0
  2884.7   0.035       0  2901.2    0.07       0  4135.9   0.045       0
  4967.5   0.045       0  5020.0   0.045       0
Bank Sta=4967.5,5020
Exp/Cntr=0.3,0.1

Type RM Length L Ch R = 1,6168,576,576,576
BEGIN DESCRIPTION:
Alkali Creek 8.0
END DESCRIPTION:
XS GIS Cut Line= 4
      1389695.77      6971257.26      1391553.44      6971055.00
      1391699.53      6971151.05      1393566.20      6970786.04
#Sta/Elev= 30
  3070.5 1930.58  3114.1 1929.57  3198.8 1929.58  3250.8 1926.50  3311.1 1926.30
  3483.3 1919.22  3532.4 1919.65  3574.7 1916.72  3633.0 1916.84  3683.3 1914.27
  3763.8 1914.70  3804.0 1912.07  3864.4 1912.88  3884.5 1910.74  4252.9 1904.79
  4427.7 1903.11  4457.9 1904.78  4494.4 1902.42  5000.8 1902.95  5007.6 1901.61
  5010.5 1896.52  5011.5 1896.02  5063.0 1896.52  5064.8 1901.78  5072.7 1902.28
  5938.7 1901.52  6739.7 1904.06  6826.5 1907.51  6892.5 1905.52  7016.0 1907.44
#Mann=6,-1,0
  3070.5   0.035       0  3114.1    0.07       0  4252.9   0.045       0
  5010.5   0.045       0  5063.0   0.045       0  6826.5    0.07       0
Bank Sta=5010.5,5063
Exp/Cntr=0.3,0.1

Type RM Length L Ch R = 1,5592,448,448,448
BEGIN DESCRIPTION:
Alkali Creek 7.0
END DESCRIPTION:
XS GIS Cut Line= 4
      1389780.91      6971314.98      1391098.15      6971416.98
      1391307.19      6971544.05      1393448.23      6971038.62
#Sta/Elev= 30
  3513.3 1930.16  3677.9 1929.66  3788.2 1922.63  3828.3 1922.63  3879.9 1919.09
  3908.6 1920.08  3958.7 1916.80  4139.8 1914.66  4189.4 1911.67  4219.5 1913.22
  4269.7 1910.03  4329.8 1910.63  4526.9 1905.56  4711.0 1902.88  4741.1 1904.49
  4801.2 1901.41  4971.2 1901.89  4979.0 1901.68  4980.1 1895.52  4981.1 1895.02
  5032.6 1895.52  5037.1 1900.87  5179.6 1902.38  6237.9 1900.82  7059.9 1904.10
  7111.3 1904.91  7121.6 1907.31  7149.1 1905.59  7217.8 1904.72  7279.0 1907.03
#Mann=5,-1,0
  3513.3    0.07       0  4526.9   0.045       0  4980.1   0.045       0
  5032.6   0.045       0  7149.1    0.07       0
Bank Sta=4980.1,5032.6
Exp/Cntr=0.3,0.1

Type RM Length L Ch R = 1,5144,630,630,630
BEGIN DESCRIPTION:
Alkali Creek 6.0
END DESCRIPTION:
XS GIS Cut Line= 4
      1389552.34      6971639.32      1391095.91      6971914.76
      1391326.43      6971926.85      1393051.15      6971497.26
#Sta/Elev= 30
  3272.7 1922.22  3404.9 1927.89  3488.7 1928.01  3748.4 1919.41  3793.5 1919.87
  3823.9 1917.15  3956.0 1913.84  3996.6 1914.72  4047.4 1911.66  4091.9 1912.67
  4118.5 1910.19  4220.1 1910.07  4263.6 1907.40  4317.5 1908.04  4395.4 1904.99
  4602.0 1902.39  4626.4 1903.84  4697.5 1901.05  4958.5 1901.61  4985.2 1900.80
  4989.9 1900.40  4993.7 1894.26  4994.7 1893.76  5046.3 1894.26  5050.0 1901.26
  5091.6 1902.03  6490.6 1900.21  6684.1 1902.84  6821.0 1905.95  6848.9 1904.45
#Mann=7,-1,0
  3272.7    0.07       0  4395.4   0.045       0  4958.5    0.07       0
  4985.2   0.045       0  4993.7   0.045       0  5046.3   0.045       0
  6684.1    0.07       0
Bank Sta=4993.7,5046.3
Exp/Cntr=0.3,0.1

Type RM Length L Ch R = 1,4514,567,567,567
BEGIN DESCRIPTION:
Alkali Creek 5.0
END DESCRIPTION:
XS GIS Cut Line= 5
      1389302.31      6972014.31      1391145.38      6972496.04
      1391286.44      6972502.55      1392300.06      6972332.69
      1393015.75      6971519.40
#Sta/Elev= 30
  3035.3 1919.90  3703.6 1917.02  3744.0 1914.14  4102.8 1912.47  4370.8 1905.87
  4629.8 1901.26  4974.7 1900.12  4990.0 1898.36  4993.7 1892.20  4994.7 1891.70
  5046.3 1892.20  5064.3 1900.73  6509.8 1900.92  6605.2 1901.93  6760.8 1895.22
  6838.6 1895.05  6874.6 1898.39  6881.3 1895.65  6895.5 1900.53  6902.2 1897.10
  6909.8 1900.40  6916.4 1896.28  6924.0 1898.87  6959.1 1895.23  6980.9 1900.09
  6987.6 1896.21  7001.8 1903.08  7036.9 1900.60  7058.7 1903.77  7192.6 1905.80
#Mann=7,-1,0
  3035.3    0.07       0  4370.8   0.045       0  4974.7    0.07       0
  4993.7    0.07       0  5046.3    0.07       0  5064.3   0.045       0
  6509.8    0.07       0
Bank Sta=4993.7,5046.3
Exp/Cntr=0.3,0.1

Type RM Length L Ch R = 1,3947,520,520,520
BEGIN DESCRIPTION:
Alkali Creek 4.0
END DESCRIPTION:
XS GIS Cut Line= 5
      1389149.58      6972257.38      1390934.30      6972981.75
      1391130.15      6973040.67      1393016.07      6972889.64
      1393264.03      6972415.34
#Sta/Elev= 30
  2947.9 1928.64  3127.1 1927.67  3288.3 1923.05  3384.2 1917.13  3413.6 1918.03
  3437.7 1915.17  3482.6 1916.11  3526.2 1912.62  3590.5 1914.22  3633.7 1910.55
  3720.0 1910.91  3741.6 1907.41  3774.0 1905.97  3942.1 1905.11  4123.5 1904.04
  4266.3 1903.22  4545.6 1902.26  4658.9 1901.68  4693.9 1903.55  4710.3 1901.89
  4950.4 1900.59  4989.6 1899.17  4990.2 1892.03  4991.2 1891.53  5042.8 1892.03
  5049.5 1898.50  5078.5 1901.06  6477.9 1898.39  7119.1 1900.84  7505.7 1903.50
#Mann=9,-1,0
  2947.9    0.07       0  3942.1   0.035       0  4123.5    0.07       0
  4266.3   0.035       0  4545.6   0.045       0  4710.3   0.035       0
  4990.2   0.035       0  5042.8   0.035       0  7119.1    0.07       0
Bank Sta=4990.2,5042.8
Exp/Cntr=0.3,0.1

Type RM Length L Ch R = 1,3427,405,405,405
BEGIN DESCRIPTION:
Alkali Creek 3.0
END DESCRIPTION:
XS GIS Cut Line= 6
      1388736.34      6972990.01      1390643.50      6973375.85
      1390905.00      6973388.00      1390980.97      6973386.76
      1393021.47      6973254.86      1393266.40      6972417.67
#Sta/Elev= 30
  2791.6 1930.47  2807.8 1931.46  2841.2 1931.63  2922.9 1927.99  3059.7 1924.15
  3218.7 1913.59  3257.5 1912.14  3320.8 1906.91  3409.7 1904.07  3414.8 1905.42
  3465.5 1902.69  3668.4 1903.75  3759.5 1902.40  4634.6 1902.02  4799.0 1901.02
  4829.0 1902.51  4887.7 1900.20  4909.1 1901.63  4933.2 1899.71  4969.2 1897.07
  4970.4 1888.81  4971.4 1888.31  5023.0 1888.81  5029.2 1899.74  5057.5 1900.40
  6852.9 1898.27  7099.8 1899.92  7751.4 1901.27  7972.8 1902.48  7992.2 1903.50
#Mann=8,-1,0
  2791.6   0.035       0  2807.8    0.07       0  4634.6   0.045       0
  4933.2    0.07       0  4970.4    0.07       0  5023.0    0.07       0
  5057.5   0.045       0  7099.8    0.07       0
Bank Sta=4970.4,5023
Exp/Cntr=0.3,0.1

Type RM Length L Ch R = 1,3022,286,286,286
BEGIN DESCRIPTION:
Alkali Creek 2.0
END DESCRIPTION:
XS GIS Cut Line= 6
      1388646.14      6973490.03      1390347.49      6973760.85
      1391118.33      6973712.24      1392968.15      6973400.19
      1393223.83      6973357.06      1393386.55      6972456.64
#Sta/Elev= 30
  2768.2 1920.26  2797.4 1920.65  2827.8 1916.16  2851.9 1916.57  3010.1 1909.71
  3100.7 1908.63  3141.7 1905.10  3202.5 1903.29  4678.9 1901.06  4718.9 1901.75
  4749.0 1904.52  4779.3 1899.13  4869.2 1896.77  4879.3 1893.67  4909.3 1897.21
  4919.3 1894.46  4928.9 1893.57  4933.9 1897.70  4939.4 1898.38  4959.4 1896.68
  4963.1 1887.37  4964.1 1886.87  5015.9 1887.37  5019.5 1896.68  5059.6 1901.93
  5517.7 1899.74  6933.3 1898.24  7141.5 1899.30  8037.8 1901.18  8313.6 1903.20
#Mann=5,-1,0
  2768.2    0.07       0  4963.1    0.07       0  5015.9    0.07       0
  5517.7   0.045       0  7141.5    0.07       0
Bank Sta=4963.1,5015.9
Exp/Cntr=0.3,0.1

Type RM Length L Ch R = 1,2736,1368,1368,1368
BEGIN DESCRIPTION:
Alkali Creek 1.0
END DESCRIPTION:
XS GIS Cut Line= 5
      1388725.95      6974444.88      1390594.34      6974246.60
      1391115.17      6973783.06      1393298.66      6973414.13
      1393475.77      6972538.31
#Sta/Elev= 30
  2772.2 1906.16  2778.3 1906.46  3847.2 1902.99  4735.3 1901.97  4799.2 1903.76
  4827.3 1902.13  4898.4 1902.08  4947.7 1900.31  4976.2 1897.15  4983.7 1894.58
  4990.4 1896.03  4992.4 1887.12  4993.4 1886.62  5045.2 1887.12  5047.2 1897.13
  5089.9 1900.67  5139.2 1902.56  5210.3 1901.12  5224.5 1902.00  5490.1 1900.21
  5527.2 1901.05  5611.8 1898.12  5642.2 1898.55  5662.5 1901.63  5682.8 1901.93
  5788.2 1898.59  7028.0 1898.23  7213.9 1899.41  8170.4 1901.41  8456.3 1903.15
#Mann=6,-1,0
  2772.2   0.035       0  2778.3    0.07       0  4992.4    0.07       0
  5045.2    0.07       0  5788.2   0.045       0  7213.9    0.07       0
Bank Sta=4992.4,5045.2
Exp/Cntr=0.3,0.1

Type RM Length L Ch R = 1,1368,331,331,331
BEGIN DESCRIPTION:
Alkali Creek 0.5
END DESCRIPTION:
XS GIS Cut Line= 5
      1390270.72      6974912.47      1391744.49      6974011.84
      1392717.38      6973988.79      1393642.98      6973434.83
      1393596.63      6972788.84
#Sta/Elev= 30
  3357.0 1903.52  4838.7 1900.67  4869.5 1900.89  4890.8 1903.35  4897.3 1901.06
  4912.1 1899.23  4927.5 1895.47  4964.3 1892.05  4965.1 1885.81  4966.1 1885.21
  5017.9 1885.81  5022.4 1894.90  5028.2 1896.83  5073.1 1900.99  5504.8 1899.92
  5654.9 1898.51  6025.0 1899.38  6077.9 1898.20  6131.2 1898.41  6225.6 1898.63
  6632.4 1898.92  6660.6 1899.20  6669.3 1900.34  6675.2 1899.42  6777.1 1899.58
  7457.9 1902.59  7714.4 1902.55  7733.0 1899.85  7738.0 1902.16  7783.7 1902.96
#Mann=5,-1,0
  3357.0    0.07       0  4965.1    0.07       0  5017.9    0.07       0
  6131.2   0.045       0  6225.6    0.07       0
Bank Sta=4965.1,5017.9
Exp/Cntr=0.3,0.1
