HEC-RAS study Buffalo Creek.prj: Buffalo Creek Base Level Engineering

--- Buffalo Creek.g01 (geometry) --- (continued)

Type RM Length L Ch R = 1,120244,404,404,404
BEGIN DESCRIPTION:
Buffalo Creek 153.0
END DESCRIPTION:
XS GIS Cut Line= 4
      1289745.66      6908589.05      1290398.43      6908007.60
      1291136.65      6907369.65      1291947.51      6906741.93
#Sta/Elev= 30
  3150.4 2371.20  3568.4 2369.17  3851.8 2362.92  3922.9 2363.33  3943.8 2360.78
  4000.7 2361.26  4113.6 2357.09  4574.3 2350.64  4575.8 2350.14  4589.6 2350.64
  5121.9 2355.14  5236.0 2359.19  5292.1 2363.68  5300.3 2362.29  5306.6 2364.29
  5314.3 2362.64  5321.1 2365.30  5335.6 2364.25  5385.4 2372.48  5742.1 2373.62
  5806.4 2374.42  5812.7 2376.75  5827.2 2374.44  5848.0 2377.11  5926.8 2375.53
  5955.8 2377.21  5976.6 2374.90  5991.1 2377.31  5997.4 2375.24  6025.7 2375.21
#Mann=3,-1,0
  3150.4    0.05       0  4574.3    0.05       0  4589.6    0.05       0
Bank Sta=4574.3,4589.6
Exp/Cntr=0.3,0.1

Type RM Length L Ch R = 1,119840,787,787,787
BEGIN DESCRIPTION:
Mapping XS caff2ccb
END DESCRIPTION:
XS GIS Cut Line= 3
      1290474.83      6908025.33      1290714.43      6907848.23
      1291589.44      6907667.68
#Sta/Elev= 30
  4149.6 2359.83  4234.1 2356.93  4269.6 2356.44  4348.8 2357.88  4473.6 2356.37
  4509.4 2353.65  4591.1 2349.67  4724.9 2351.54  4770.1 2350.15  4799.3 2350.11
  4865.5 2349.63  4920.9 2351.33  4963.8 2349.06  4971.1 2349.54  4979.1 2348.96
  4981.6 2348.00  4983.1 2347.50  4996.9 2348.00  4999.5 2349.65  5009.7 2350.74
  5050.6 2353.64  5066.6 2355.65  5116.8 2358.42  5132.2 2360.86  5173.1 2360.86
  5212.3 2363.65  5244.6 2363.70  5275.2 2365.04  5305.8 2367.71  5341.0 2367.39
#Mann=5,-1,0
  4149.6    0.05       0  4799.3    0.12       0  4963.8    0.05       0
  4981.6    0.05       0  4996.9    0.05       0
Bank Sta=4981.6,4996.9
Exp/Cntr=0.3,0.1

Type RM Length L Ch R = 1,119053,308,308,308
BEGIN DESCRIPTION:
Mapping XS 54e9c5d2
END DESCRIPTION:
XS GIS Cut Line= 2
      1291016.50      6908573.95      1291488.71      6907945.49
#Sta/Elev= 30
  4642.7 2361.61  4767.0 2357.79  4860.7 2353.43  4902.4 2352.88  4968.5 2348.04
  4975.3 2347.18  5002.4 2346.31  5023.8 2344.92  5025.3 2344.42  5037.7 2344.42
  5039.2 2344.92  5046.1 2346.53  5060.7 2346.46  5075.3 2347.53  5110.7 2348.96
  5131.5 2348.90  5159.1 2350.53  5175.2 2352.27  5196.1 2352.12  5231.5 2354.55
  5246.1 2354.83  5252.3 2355.53  5260.6 2355.33  5266.9 2356.29  5275.2 2356.00
  5281.5 2356.85  5310.6 2357.93  5316.9 2358.97  5366.9 2358.57  5428.8 2359.59
#Mann=5,-1,0
  4642.7    0.05       0  4968.5    0.12       0  5023.8    0.07       0
  5039.2    0.12       0  5159.1    0.05       0
Bank Sta=5023.8,5039.2
Exp/Cntr=0.3,0.1

Type RM Length L Ch R = 1,118745,363,363,363
BEGIN DESCRIPTION:
Buffalo Creek 150.0
END DESCRIPTION:
XS GIS Cut Line= 3
      1291054.98      6909038.04      1291455.00      6908438.00
      1291855.04      6908137.97
#Sta/Elev= 30
  4274.3 2369.06  4296.9 2367.11  4549.3 2361.85  4627.4 2359.26  4663.4 2360.40
  4684.5 2358.29  4714.5 2357.81  4771.6 2354.78  4786.6 2354.99  4792.6 2353.94
  4801.7 2354.07  4807.7 2352.93  4828.7 2351.93  4858.7 2351.50  4879.8 2349.59
  4981.9 2345.88  4995.0 2342.94  4996.5 2342.44  5010.4 2342.94  5031.9 2344.37
  5038.2 2345.87  5081.9 2348.04  5131.9 2352.92  5281.9 2361.80  5388.2 2366.15
  5402.7 2365.36  5438.2 2367.01  5488.2 2367.30  5492.3 2368.69  5495.5 2368.69
#Mann=3,-1,0
  4274.3    0.05       0  4995.0    0.05       0  5010.4    0.05       0
Bank Sta=4995,5010.4
Exp/Cntr=0.3,0.1

Type RM Length L Ch R = 1,118382,176,176,176
BEGIN DESCRIPTION:
Buffalo Creek 149.0
END DESCRIPTION:
XS GIS Cut Line= 3
      1291393.23      6909422.27      1291602.31      6908760.05
      1291769.58      6908211.74
#Sta/Elev= 30
  4286.3 2368.16  4322.2 2369.22  4377.6 2366.25  4552.9 2362.01  4609.2 2361.87
  4641.5 2359.57  4668.3 2356.20  4699.8 2357.19  4808.4 2353.37  4835.5 2351.31
  4846.6 2349.21  4905.4 2345.48  4930.5 2345.30  4967.6 2342.14  4969.1 2341.64
  4983.1 2342.14  4984.4 2343.54  4993.3 2345.19  5035.2 2346.14  5087.4 2349.28
  5192.0 2351.55  5417.6 2360.70  5422.8 2360.14  5450.4 2361.84  5455.6 2360.79
  5483.2 2362.96  5488.4 2361.91  5516.0 2363.65  5521.3 2362.93  5554.0 2365.59
#Mann=3,-1,0
  4286.3    0.05       0  4967.6    0.05       0  4983.1    0.05       0
Bank Sta=4967.6,4983.1
Exp/Cntr=0.3,0.1

Type RM Length L Ch R = 1,118206,562,562,562
BEGIN DESCRIPTION:
Buffalo Creek 149.5
END DESCRIPTION:
XS GIS Cut Line= 2
      1291613.35      6909416.49      1291904.32      6908193.42
#Sta/Elev= 30
  4398.9 2362.82  4509.7 2361.68  4572.1 2360.25  4654.3 2357.14  4767.4 2354.28
  4829.1 2351.24  4862.4 2349.08  4880.5 2347.08  4899.4 2346.72  4952.4 2343.29
  4983.3 2342.29  4994.0 2341.21  5003.8 2341.40  5006.3 2339.96  5007.8 2339.46
  5020.3 2339.46  5021.8 2339.96  5024.4 2341.38  5044.9 2343.48  5106.6 2346.67
  5199.1 2349.85  5240.2 2352.09  5247.0 2353.15  5289.1 2356.12  5468.1 2363.52
  5552.4 2366.40  5558.9 2365.97  5594.6 2368.13  5620.6 2367.98  5656.1 2369.03
#Mann=3,-1,0
  4398.9    0.05       0  5006.3   0.033       0  5021.8    0.05       0
Bank Sta=5006.3,5021.8
Exp/Cntr=0.3,0.1

Type RM Length L Ch R = 1,117644,542,542,542
BEGIN DESCRIPTION:
Buffalo Creek 148.0
END DESCRIPTION:
XS GIS Cut Line= 3
      1291500.29      6909861.20      1292255.00      6909038.00
      1292454.99      6908688.02
#Sta/Elev= 30
  3890.4 2370.47  4080.1 2366.11  4334.8 2357.96  4596.8 2353.30  4731.3 2348.31
  4766.4 2345.94  4816.4 2345.11  4844.4 2342.76  4858.3 2340.06  4936.6 2339.09
  4943.4 2337.47  4978.2 2335.65  4979.7 2335.15  4993.7 2335.65  5003.8 2338.13
  5015.1 2338.68  5020.9 2342.14  5030.2 2341.93  5036.7 2345.02  5042.5 2346.58
  5052.6 2347.14  5058.3 2349.34  5074.2 2349.91  5079.9 2350.99  5095.7 2350.49
  5101.5 2351.87  5203.7 2357.50  5262.8 2359.11  5352.7 2363.52  5410.3 2364.88
#Mann=3,-1,0
  3890.4    0.05       0  4978.2    0.05       0  4993.7    0.05       0
Bank Sta=4978.2,4993.7
Exp/Cntr=0.3,0.1

Type RM Length L Ch R = 1,117102,549,549,549
BEGIN DESCRIPTION:
Buffalo Creek 147.0
END DESCRIPTION:
XS GIS Cut Line= 3
      1292104.99      6909938.02      1292505.00      6909488.00
      1292775.50      6908948.96
#Sta/Elev= 30
  4398.4 2359.40  4490.8 2358.40  4611.2 2355.48  4766.8 2349.95  4858.8 2345.29
  4915.6 2343.67  4944.1 2339.87  4950.7 2336.96  4958.3 2334.90  4962.9 2334.60
  4964.7 2332.63  4966.2 2332.13  4980.3 2332.63  5003.3 2334.27  5014.5 2336.17
  5036.8 2336.54  5053.5 2338.22  5142.9 2344.06  5165.2 2344.26  5170.8 2343.68
  5187.6 2344.53  5193.2 2344.00  5304.8 2347.71  5321.6 2349.81  5438.9 2354.65
  5483.5 2358.02  5505.9 2358.85  5515.2 2360.19  5528.2 2360.14  5603.6 2364.01
#Mann=3,-1,0
  4398.4    0.05       0  4964.7    0.05       0  4980.3    0.05       0
Bank Sta=4964.7,4980.3
Exp/Cntr=0.3,0.1

Type RM Length L Ch R = 1,116553,549,549,549
BEGIN DESCRIPTION:
Buffalo Creek 146.0
END DESCRIPTION:
XS GIS Cut Line= 3
      1292255.05      6909937.99      1292655.00      6909888.00
      1293153.19      6909702.71
#Sta/Elev= 30
  4591.0 2357.25  4714.4 2352.71  4772.4 2349.53  4832.8 2344.85  4842.9 2344.64
  4875.7 2341.79  4903.4 2338.76  4943.7 2335.76  4963.8 2332.50  4973.9 2329.86
  4976.2 2328.59  4977.7 2328.09  4990.3 2328.09  4991.8 2328.59  5015.4 2329.98
  5034.3 2333.76  5039.6 2333.50  5064.6 2339.35  5069.9 2338.64  5089.6 2339.25
  5100.8 2339.08  5120.0 2342.40  5132.8 2343.73  5155.6 2344.33  5241.3 2348.83
  5296.7 2350.87  5367.5 2354.30  5431.5 2357.92  5443.1 2358.97  5525.6 2362.32
#Mann=3,-1,0
  4591.0    0.05       0  4976.2    0.05       0  4991.8    0.05       0
Bank Sta=4976.2,4991.8
Exp/Cntr=0.3,0.1

Type RM Length L Ch R = 1,116004,569,569,569
BEGIN DESCRIPTION:
Buffalo Creek 145.0
END DESCRIPTION:
XS GIS Cut Line= 3
      1292654.99      6910488.01      1293005.00      6910188.00
      1293205.00      6909838.00
#Sta/Elev= 30
  4534.3 2355.53  4640.2 2352.88  4754.4 2346.10  4789.5 2344.79  4846.6 2340.55
  4881.7 2338.97  4896.0 2337.23  4916.8 2337.27  4959.6 2334.23  4967.3 2332.30
  4981.6 2330.82  4998.2 2330.19  5003.2 2329.32  5009.0 2325.55  5010.5 2323.51
  5012.0 2323.01  5026.1 2323.51  5040.6 2327.42  5046.4 2330.28  5062.2 2334.03
  5068.0 2338.16  5098.9 2337.53  5121.3 2339.93  5148.6 2345.13  5164.5 2346.64
  5229.2 2348.02  5245.1 2349.69  5250.8 2349.01  5309.9 2354.61  5398.4 2359.81
#Mann=3,-1,0
  4534.3    0.05       0  5010.5   0.033       0  5026.1    0.05       0
Bank Sta=5010.5,5026.1
Exp/Cntr=0.3,0.1

Type RM Length L Ch R = 1,115435,545,545,545
BEGIN DESCRIPTION:
Buffalo Creek 144.0
END DESCRIPTION:
XS GIS Cut Line= 3
      1292755.02      6910738.00      1293155.00      6910688.00
      1293505.00      6910488.00
#Sta/Elev= 30
  4592.3 2354.47  4715.7 2349.85  4723.3 2348.84  4791.3 2344.22  4796.4 2344.43
  4894.6 2337.74  4904.7 2335.69  4952.6 2329.26  4957.6 2326.36  4975.2 2322.87
  4977.5 2321.57  4979.0 2321.07  4991.7 2321.07  4993.2 2321.57  4995.4 2322.87
  4998.3 2322.87  5003.3 2324.50  5009.1 2323.25  5018.4 2326.79  5024.9 2328.27
  5030.7 2327.16  5046.5 2330.23  5053.0 2332.08  5099.1 2336.55  5111.3 2338.44
  5127.1 2338.77  5143.0 2340.86  5170.3 2342.24  5214.2 2346.36  5398.5 2357.77
#Mann=3,-1,0
  4592.3    0.05       0  4977.5   0.033       0  4993.2    0.05       0
Bank Sta=4977.5,4993.2
Exp/Cntr=0.3,0.1

Type RM Length L Ch R = 1,114890,602,602,602
BEGIN DESCRIPTION:
Buffalo Creek 143.0
END DESCRIPTION:
XS GIS Cut Line= 3
      1293055.03      6911138.00      1293455.00      6911088.00
      1293805.01      6910888.00
#Sta/Elev= 30
  4596.7 2353.24  4768.0 2350.02  4788.1 2348.82  4800.7 2344.17  4808.3 2342.40
  4818.4 2341.06  4868.8 2337.59  4919.2 2332.50  4957.0 2324.50  4962.0 2324.75
  4979.6 2322.93  4989.4 2320.14  4990.9 2319.64  5005.1 2320.14  5013.5 2320.42
  5022.8 2322.01  5035.1 2327.71  5045.1 2325.86  5057.4 2329.23  5066.7 2333.35
  5080.4 2335.13  5088.3 2337.10  5161.0 2341.94  5190.5 2344.81  5218.6 2349.02
  5255.3 2352.06  5264.7 2352.00  5276.9 2354.53  5322.3 2356.77  5402.9 2357.70
#Mann=3,-1,0
  4596.7    0.05       0  4989.4   0.033       0  5005.1    0.05       0
Bank Sta=4989.4,5005.1
Exp/Cntr=0.3,0.1

Type RM Length L Ch R = 1,114288,640,640,640
BEGIN DESCRIPTION:
Buffalo Creek 142.0
END DESCRIPTION:
XS GIS Cut Line= 3
      1293388.42      6911665.28      1293756.45      6911561.11
      1294104.96      6911438.01
#Sta/Elev= 30
  4619.3 2346.52  4761.2 2340.28  4887.9 2332.77  4916.7 2329.90  4921.9 2328.54
  4937.9 2325.99  4961.0 2323.78  4969.1 2320.86  4971.6 2317.88  4973.1 2317.38
  4985.9 2317.38  4987.4 2317.88  4989.8 2320.02  4995.0 2320.54  4998.4 2323.76
  5010.9 2324.70  5021.2 2326.33  5026.5 2326.28  5032.1 2328.55  5106.3 2332.24
  5119.2 2333.55  5138.1 2333.86  5201.4 2337.24  5212.4 2338.34  5254.8 2340.16
  5263.2 2341.52  5268.5 2341.57  5307.8 2345.11  5325.1 2347.68  5371.4 2350.23
#Mann=3,-1,0
  4619.3    0.05       0  4971.6    0.05       0  4987.4    0.05       0
Bank Sta=4971.6,4987.4
Exp/Cntr=0.3,0.1

Type RM Length L Ch R = 1,113648,400,400,400
BEGIN DESCRIPTION:
Buffalo Creek 141.0
END DESCRIPTION:
XS GIS Cut Line= 3
      1293518.55      6912337.84      1294030.41      6911990.59
      1294344.94      6911563.55
#Sta/Elev= 30
  4397.9 2350.55  4439.0 2350.08  4460.0 2348.65  4475.0 2348.63  4502.4 2347.13
  4561.8 2345.68  4654.7 2341.49  4675.6 2339.85  4705.5 2339.03  4768.5 2335.64
  4828.3 2331.32  4885.2 2328.87  4913.2 2327.01  4936.1 2323.73  4985.7 2321.06
  4999.1 2318.75  5006.1 2315.13  5007.6 2314.63  5022.0 2315.13  5029.2 2320.02
  5035.4 2321.75  5043.9 2322.32  5064.7 2325.58  5085.6 2327.77  5150.3 2331.91
  5215.1 2334.84  5365.5 2344.43  5401.0 2347.46  5486.6 2352.22  5546.8 2354.70
#Mann=3,-1,0
  4397.9    0.05       0  5006.1    0.05       0  5022.0    0.05       0
Bank Sta=5006.1,5022
Exp/Cntr=0.3,0.1

Type RM Length L Ch R = 1,113248,531,531,531
BEGIN DESCRIPTION:
Buffalo Creek 140.0
END DESCRIPTION:
XS GIS Cut Line= 3
      1293855.04      6912537.98      1294205.00      6912338.00
      1294555.01      6911937.98
#Sta/Elev= 30
  4591.7 2350.00  4658.6 2347.08  4782.4 2337.65  4804.0 2336.85  4819.8 2334.95
  4825.6 2335.06  4847.2 2331.56  4878.9 2328.44  4922.1 2327.68  4937.2 2326.47
  4943.7 2324.31  4949.4 2320.57  4959.5 2318.69  4971.7 2318.10  4986.9 2315.58
  5000.6 2315.04  5002.1 2314.54  5016.5 2315.04  5022.8 2320.92  5030.4 2323.35
  5079.7 2322.95  5129.1 2324.94  5171.8 2324.38  5179.4 2326.17  5186.0 2326.58
  5412.9 2339.00  5448.0 2341.86  5469.8 2347.28  5476.4 2347.78  5526.3 2348.94
#Mann=3,-1,0
  4591.7    0.05       0  5000.6   0.033       0  5016.5    0.05       0
Bank Sta=5000.6,5016.5
Exp/Cntr=0.3,0.1

Type RM Length L Ch R = 1,112717,622,622,622
BEGIN DESCRIPTION:
Buffalo Creek 139.0
END DESCRIPTION:
XS GIS Cut Line= 3
      1294202.60      6912990.60      1294505.00      6912688.00
      1294854.99      6912488.01
#Sta/Elev= 30
  4577.3 2344.05  4616.2 2342.18  4750.5 2332.45  4778.8 2327.78  4807.1 2326.21
  4842.5 2321.85  4877.8 2321.31  4913.2 2322.18  4955.6 2318.29  4962.7 2318.62
  4976.8 2316.26  4983.0 2310.91  4984.5 2310.41  4999.0 2310.91  5001.6 2316.01
  5008.0 2316.01  5018.8 2318.36  5062.7 2318.97  5115.2 2324.09  5158.4 2326.25
  5180.0 2325.81  5195.9 2324.12  5211.7 2324.44  5239.1 2325.34  5292.3 2329.54
  5313.9 2333.05  5335.5 2337.98  5357.1 2340.76  5362.9 2342.60  5408.2 2345.47
#Mann=3,-1,0
  4577.3    0.05       0  4983.0   0.033       0  4999.0    0.05       0
Bank Sta=4983,4999
Exp/Cntr=0.3,0.1

Type RM Length L Ch R = 1,112095,384,384,384
BEGIN DESCRIPTION:
Buffalo Creek 138.0
END DESCRIPTION:
XS GIS Cut Line= 3
      1294355.04      6913187.99      1294717.91      6913073.93
      1295104.97      6912938.01
#Sta/Elev= 30
  4601.9 2346.30  4664.8 2347.79  4688.1 2347.32  4720.5 2345.95  4752.9 2342.94
  4790.5 2332.04  4832.5 2326.04  4855.3 2318.09  4887.7 2315.97  4905.8 2316.35
  4914.9 2315.31  4937.3 2315.25  4952.5 2313.27  4968.7 2315.08  4976.8 2308.18
  4978.3 2307.68  4992.8 2308.18  5000.4 2313.82  5032.2 2317.47  5041.5 2317.42
  5046.8 2319.14  5072.4 2319.29  5170.7 2328.59  5196.4 2332.65  5201.8 2335.43
  5222.1 2341.46  5233.6 2344.52  5244.2 2345.79  5284.1 2347.51  5392.5 2349.32
#Mann=3,-1,0
  4601.9    0.05       0  4976.8    0.05       0  4992.8    0.05       0
Bank Sta=4976.8,4992.8
Exp/Cntr=0.3,0.1

Type RM Length L Ch R = 1,111711,624,624,624
BEGIN DESCRIPTION:
Buffalo Creek 137.0
END DESCRIPTION:
XS GIS Cut Line= 3
      1294285.95      6913417.69      1294971.38      6913310.04
      1295470.65      6913171.35
#Sta/Elev= 30
  4322.5 2344.34  4417.4 2340.95  4480.0 2337.38  4493.6 2337.31  4635.3 2328.19
  4677.9 2325.00  4685.9 2323.82  4746.7 2319.64  4808.2 2318.49  4817.5 2317.79
  4847.9 2318.40  4878.3 2317.19  4908.6 2314.93  4949.1 2314.75  4969.4 2311.26
  4979.5 2310.57  4981.6 2307.85  4983.1 2307.35  4997.6 2307.85  5001.0 2309.55
  5009.9 2317.12  5015.6 2320.39  5020.8 2320.39  5030.5 2323.46  5039.1 2325.22
  5051.2 2326.26  5157.5 2333.19  5339.1 2342.37  5344.3 2343.14  5534.5 2350.84
#Mann=3,-1,0
  4322.5    0.05       0  4981.6    0.05       0  4997.6    0.05       0
Bank Sta=4981.6,4997.6
Exp/Cntr=0.3,0.1

Type RM Length L Ch R = 1,111087,373,373,373
BEGIN DESCRIPTION:
Buffalo Creek 136.0
END DESCRIPTION:
XS GIS Cut Line= 3
      1294179.96      6913813.00      1294755.00      6913838.00
      1295260.81      6913841.30
#Sta/Elev= 30
  4424.8 2348.10  4499.9 2346.77  4519.9 2345.49  4570.0 2343.83  4600.0 2342.24
  4640.0 2339.40  4670.1 2338.06  4680.1 2336.86  4720.1 2333.96  4810.2 2328.97
  4840.2 2326.37  4930.3 2320.23  4940.3 2319.20  4960.3 2315.82  4970.4 2314.98
  4980.4 2312.18  4989.9 2305.66  4991.4 2305.16  5004.4 2305.16  5005.9 2305.66
  5010.4 2309.92  5020.4 2311.63  5040.4 2312.23  5060.4 2314.74  5070.4 2313.73
  5110.4 2315.36  5290.4 2325.14  5400.4 2330.35  5500.4 2334.24  5506.2 2334.90
#Mann=3,-1,0
  4424.8    0.05       0  4989.9    0.05       0  5005.9    0.05       0
Bank Sta=4989.9,5005.9
Exp/Cntr=0.3,0.1

Type RM Length L Ch R = 1,110714,1212,1212,1212
BEGIN DESCRIPTION:
Buffalo Creek 135.5
END DESCRIPTION:
XS GIS Cut Line= 3
      1294336.68      6914119.49      1294742.42      6914212.70
      1295389.48      6914108.51
#Sta/Elev= 30
  4571.0 2341.95  4633.7 2341.35  4676.5 2339.62  4719.4 2335.79  4724.5 2336.32
  4762.2 2332.95  4810.2 2330.42  4825.8 2328.66  4836.1 2324.99  4853.0 2322.38
  4901.0 2317.58  4943.9 2311.96  4949.0 2312.30  4959.2 2310.97  4969.4 2307.13
  4971.7 2305.25  4973.2 2304.75  4987.7 2305.25  4991.1 2307.30  5010.2 2310.68
  5091.2 2310.24  5108.8 2307.06  5113.9 2308.39  5141.9 2310.84  5192.5 2312.94
  5222.9 2316.66  5273.5 2317.32  5293.8 2318.35  5304.5 2319.95  5642.7 2334.36
#Mann=3,-1,0
  4571.0    0.05       0  4971.7    0.05       0  4987.7    0.05       0
Bank Sta=4971.7,4987.7
Exp/Cntr=0.3,0.1

Type RM Length L Ch R = 1,109502,653,653,653
BEGIN DESCRIPTION:
Buffalo Creek 135.0
END DESCRIPTION:
XS GIS Cut Line= 4
      1294318.62      6914435.06      1294830.00      6914813.00
      1294905.00      6914788.00      1295454.97      6914638.01
#Sta/Elev= 30
  4285.0 2334.11  4399.0 2333.54  4549.3 2324.22  4584.8 2320.64  4720.5 2313.00
  4820.7 2310.70  4968.3 2310.56  5022.4 2301.43  5051.8 2303.16  5062.1 2306.21
  5124.3 2304.45  5131.2 2302.50  5136.4 2305.59  5145.1 2304.35  5155.4 2300.11
  5168.1 2299.68  5169.6 2299.18  5184.1 2299.68  5186.5 2301.19  5205.5 2302.58
  5210.7 2306.10  5300.5 2309.25  5342.0 2314.41  5359.3 2314.98  5373.1 2317.83
  5383.5 2317.19  5393.8 2318.44  5404.2 2323.83  5414.6 2325.15  5570.0 2335.97
#Mann=3,-1,0
  4285.0    0.05       0  5168.1    0.05       0  5184.1    0.05       0
Bank Sta=5168.1,5184.1
Exp/Cntr=0.3,0.1

Type RM Length L Ch R = 1,108849,421,421,421
BEGIN DESCRIPTION:
Buffalo Creek 134.0
END DESCRIPTION:
XS GIS Cut Line= 3
      1294463.73      6915555.81      1295074.91      6915291.95
      1295405.02      6914887.98
#Sta/Elev= 30
  4410.4 2330.01  4446.3 2328.50  4575.2 2319.07  4598.2 2318.62  4744.7 2309.99
  4814.8 2308.44  4925.6 2307.93  4934.6 2305.29  4943.7 2299.64  4948.4 2294.71
  4949.9 2294.21  4964.4 2294.71  4967.2 2296.99  4972.6 2298.02  4978.2 2299.00
  4996.1 2299.37  5001.6 2301.47  5093.8 2303.78  5164.2 2309.51  5207.2 2310.81
  5335.0 2317.28  5384.6 2321.12  5398.9 2321.08  5405.4 2322.05  5434.1 2323.56
  5442.0 2323.23  5448.4 2324.15  5520.2 2325.47  5561.9 2328.61  5597.8 2330.07
#Mann=3,-1,0
  4410.4    0.05       0  4948.4    0.05       0  4964.4    0.05       0
Bank Sta=4948.4,4964.4
Exp/Cntr=0.3,0.1

Type RM Length L Ch R = 1,108428,688,688,688
BEGIN DESCRIPTION:
Buffalo Creek 133.0
END DESCRIPTION:
XS GIS Cut Line= 3
      1294446.02      6915830.54      1295155.00      6915688.00
      1295919.97      6915554.50
#Sta/Elev= 30
  4272.9 2332.19  4353.5 2327.02  4475.9 2317.54  4537.1 2313.94  4716.3 2308.42
  4802.3 2306.97  4924.9 2306.26  4945.1 2305.39  4955.3 2301.27  4962.6 2294.38
  4964.1 2293.88  4978.6 2294.38  4985.9 2296.65  5006.2 2296.58  5023.3 2297.81
  5028.4 2300.15  5077.3 2301.70  5087.9 2304.09  5107.7 2306.92  5117.9 2307.61
  5142.4 2308.39  5188.9 2307.99  5256.4 2309.58  5270.1 2308.90  5392.0 2313.36
  5442.7 2314.22  5543.9 2317.44  5716.8 2323.61  5722.5 2324.32  5772.6 2325.41
#Mann=3,-1,0
  4272.9    0.05       0  4962.6    0.05       0  4978.6    0.05       0
Bank Sta=4962.6,4978.6
Exp/Cntr=0.3,0.1

Type RM Length L Ch R = 1,107740,953,953,953
BEGIN DESCRIPTION:
Mapping XS 453d3822
END DESCRIPTION:
XS GIS Cut Line= 3
      1295210.96      6916448.93      1295540.82      6916042.68
      1295873.84      6915612.53
#Sta/Elev= 30
  4292.9 2314.96  4318.3 2313.75  4324.7 2312.64  4423.8 2308.07  4446.1 2306.22
  4658.7 2303.09  4693.9 2299.70  4722.7 2298.60  4737.0 2298.61  4751.4 2300.47
  4786.6 2298.93  4829.8 2300.31  4836.1 2299.63  4867.3 2299.60  4914.9 2297.02
  4943.9 2297.84  4964.7 2295.44  4993.7 2295.31  5006.5 2291.71  5008.0 2291.21
  5022.5 2291.71  5029.0 2294.27  5037.1 2301.88  5043.5 2309.87  5049.8 2312.41
  5087.0 2314.48  5100.4 2313.35  5146.3 2314.05  5286.2 2317.46  5360.2 2322.68
#Mann=5,-1,0
  4292.9    0.05       0  4867.3    0.12       0  5006.5    0.07       0
  5022.5    0.12       0  5146.3    0.05       0
Bank Sta=5006.5,5022.5
Exp/Cntr=0.3,0.1

Type RM Length L Ch R = 1,106787,531,531,531
BEGIN DESCRIPTION:
Buffalo Creek 131.0
END DESCRIPTION:
XS GIS Cut Line= 3
      1295504.99      6916888.01      1295855.00      6916288.00
      1296504.98      6915688.02
#Sta/Elev= 30
  4303.9 2333.27  4311.8 2331.80  4589.6 2313.49  4616.9 2312.62  4669.8 2308.12
  4755.8 2303.67  4812.2 2302.10  4830.3 2301.67  4846.0 2299.32  4851.8 2299.54
  4859.6 2297.69  4889.0 2294.32  4894.8 2294.72  4963.4 2289.27  4969.2 2289.98
  4982.7 2286.72  4984.2 2286.22  4998.7 2286.72  5001.9 2290.84  5005.6 2287.93
  5012.4 2292.45  5019.8 2291.47  5026.6 2298.63  5034.0 2295.61  5040.8 2302.10
  5157.4 2304.02  5310.1 2305.63  5472.9 2313.01  5564.7 2318.30  5883.1 2340.48
#Mann=5,-1,0
  4303.9    0.05       0  4812.2    0.12       0  4982.7    0.07       0
  4998.7    0.12       0  5157.4    0.05       0
Bank Sta=4982.7,4998.7
Exp/Cntr=0.3,0.1

Type RM Length L Ch R = 1,106256,572,572,572
BEGIN DESCRIPTION:
Buffalo Creek 130.0
END DESCRIPTION:
XS GIS Cut Line= 3
      1295705.00      6917038.00      1296255.00      6916588.00
      1296705.00      6915888.00
#Sta/Elev= 30
  4284.6 2332.18  4483.4 2316.98  4576.0 2310.90  4582.5 2311.24  4683.0 2305.13
  4775.6 2302.24  4860.3 2298.20  4866.7 2296.75  4889.0 2295.50  4930.6 2294.95
  4963.8 2293.03  5002.8 2289.21  5016.0 2285.68  5017.5 2285.18  5032.0 2285.68
  5039.2 2292.96  5045.1 2296.08  5054.3 2299.04  5060.3 2295.52  5066.6 2299.78
  5162.8 2300.51  5278.2 2300.52  5350.9 2302.27  5387.2 2304.16  5429.5 2306.78
  5502.1 2313.28  5517.3 2313.67  5565.9 2318.40  5574.8 2318.33  5827.4 2339.53
#Mann=5,-1,0
  4284.6    0.05       0  4963.8    0.12       0  5016.0    0.07       0
  5032.0    0.12       0  5162.8    0.05       0
Bank Sta=5016,5032
Exp/Cntr=0.3,0.1

Type RM Length L Ch R = 1,105684,548,548,548
BEGIN DESCRIPTION:
Buffalo Creek 129.0
END DESCRIPTION:
XS GIS Cut Line= 3
      1295704.99      6917088.00      1296455.00      6917038.00
      1297204.98      6916938.00
#Sta/Elev= 30
  4252.2 2332.86  4362.5 2325.70  4492.7 2315.10  4572.9 2310.78  4703.2 2302.00
  4753.3 2300.09  4773.4 2298.58  4833.5 2296.83  4933.7 2296.47  4953.8 2290.27
  4965.8 2282.86  4967.3 2282.36  4981.8 2282.86  5006.4 2283.99  5014.0 2285.89
  5034.1 2287.63  5040.4 2290.44  5045.5 2290.87  5054.3 2293.92  5074.5 2296.08
  5215.7 2297.44  5336.8 2301.93  5343.1 2303.16  5387.2 2304.67  5457.9 2309.39
  5518.4 2314.11  5528.5 2315.64  5538.6 2315.67  5558.7 2318.03  5760.5 2331.71
#Mann=3,-1,0
  4252.2    0.05       0  4965.8    0.05       0  4981.8    0.05       0
Bank Sta=4965.8,4981.8
Exp/Cntr=0.3,0.1

Type RM Length L Ch R = 1,105136,557,557,557
BEGIN DESCRIPTION:
Buffalo Creek 128.0
END DESCRIPTION:
XS GIS Cut Line= 4
      1295674.46      6917790.75      1296453.49      6917488.50
      1296507.77      6917365.41      1297261.52      6917096.83
#Sta/Elev= 30
  4164.4 2330.71  4267.8 2325.53  4412.0 2316.54  4624.5 2306.30  4690.6 2304.20
  4787.1 2303.26  4926.5 2300.07  4932.1 2299.67  4937.5 2291.41  4956.6 2287.47
  4962.0 2284.38  4978.6 2282.04  4980.1 2281.54  4994.6 2282.04  4998.1 2284.12
  5003.0 2284.12  5011.1 2286.52  5016.5 2286.16  5039.9 2290.83  5092.0 2290.24
  5115.3 2291.43  5144.6 2295.69  5375.3 2294.28  5428.8 2295.98  5460.7 2298.71
  5560.2 2304.13  5598.7 2308.25  5709.0 2315.28  5796.1 2322.56  5934.7 2330.81
#Mann=3,-1,0
  4164.4    0.05       0  4978.6    0.05       0  4994.6    0.05       0
Bank Sta=4978.6,4994.6
Exp/Cntr=0.3,0.1

Type RM Length L Ch R = 1,104579,562,562,562
BEGIN DESCRIPTION:
Buffalo Creek 127.0
END DESCRIPTION:
XS GIS Cut Line= 3
      1296504.99      6918488.02      1296855.00      6917688.00
      1297155.00      6917388.00
#Sta/Elev= 30
  4126.8 2318.94  4287.0 2309.24  4292.5 2309.70  4301.5 2308.43  4414.9 2302.87
  4421.5 2301.72  4443.7 2300.20  4454.3 2300.22  4584.1 2293.45  4787.6 2292.44
  4811.0 2293.06  4816.4 2292.40  4910.0 2293.14  4938.8 2289.21  4978.2 2288.18
  4985.6 2286.71  4989.3 2279.04  4990.8 2278.54  5005.3 2279.04  5014.2 2283.11
  5070.7 2287.12  5084.9 2286.90  5099.0 2288.43  5113.2 2291.40  5141.5 2295.38
  5155.6 2295.37  5226.3 2300.02  5268.7 2303.84  5367.7 2315.17  5424.3 2318.70
#Mann=3,-1,0
  4126.8    0.05       0  4989.3    0.05       0  5005.3    0.05       0
Bank Sta=4989.3,5005.3
Exp/Cntr=0.3,0.1

Type RM Length L Ch R = 1,104017,553,553,553
BEGIN DESCRIPTION:
Buffalo Creek 126.0
END DESCRIPTION:
XS GIS Cut Line= 3
      1296605.03      6918787.96      1297155.00      6918038.00
      1297492.64      6917262.09
#Sta/Elev= 30
  4075.3 2335.75  4153.6 2330.33  4174.5 2326.04  4189.1 2327.62  4440.0 2307.72
  4454.6 2305.43  4569.6 2297.63  4761.8 2290.23  4897.6 2290.71  4933.2 2284.19
  4962.5 2282.26  4969.1 2276.11  4970.6 2275.61  4985.1 2276.11  4998.0 2284.08
  5008.0 2285.42  5019.8 2290.37  5103.5 2289.48  5125.3 2286.72  5189.3 2287.86
  5223.6 2291.40  5293.9 2292.14  5322.8 2296.48  5376.1 2298.00  5573.5 2308.74
  5591.5 2310.75  5620.4 2310.71  5649.3 2313.31  5795.4 2319.82  5851.5 2324.10
#Mann=3,-1,0
  4075.3    0.05       0  4969.1    0.05       0  4985.1    0.05       0
Bank Sta=4969.1,4985.1
Exp/Cntr=0.3,0.1

Type RM Length L Ch R = 1,103464,508,508,508
BEGIN DESCRIPTION:
Buffalo Creek 125.0
END DESCRIPTION:
XS GIS Cut Line= 3
      1296705.01      6918937.99      1297505.00      6918138.00
      1298130.54      6917556.84
#Sta/Elev= 30
  3869.1 2337.01  4024.7 2327.14  4052.9 2324.86  4081.2 2320.18  4095.4 2322.64
  4392.3 2305.78  4406.5 2305.98  4576.2 2297.86  4745.9 2291.70  4788.3 2289.29
  4859.0 2286.81  4929.8 2287.35  4943.9 2284.61  4958.0 2278.79  4964.2 2274.08
  4965.7 2273.58  4980.2 2274.08  4986.3 2280.61  4996.9 2282.43  5014.4 2282.77
  5056.9 2287.12  5219.6 2296.77  5403.8 2305.43  5503.0 2312.33  5651.5 2325.40
  5708.2 2328.17  5757.6 2328.60  5771.7 2330.15  5778.6 2329.17  5854.3 2328.90
#Mann=3,-1,0
  3869.1    0.05       0  4964.2    0.05       0  4980.2    0.05       0
Bank Sta=4964.2,4980.2
Exp/Cntr=0.3,0.1

Type RM Length L Ch R = 1,102956,566,566,566
BEGIN DESCRIPTION:
Buffalo Creek 124.0
END DESCRIPTION:
XS GIS Cut Line= 3
      1297154.99      6919188.01      1297905.00      6918388.00
      1298205.01      6917687.98
#Sta/Elev= 30
  3898.9 2333.18  3927.0 2330.49  4125.3 2318.31  4146.3 2316.35  4153.6 2313.57
  4174.7 2315.28  4302.1 2306.50  4528.8 2294.92  4790.1 2286.99  4945.9 2285.97
  4960.1 2284.29  4967.4 2282.05  4988.4 2280.45  4992.1 2273.23  4995.5 2273.23
  4996.6 2271.72  4998.1 2271.22  5012.6 2271.72  5017.3 2275.36  5039.0 2283.90
  5057.2 2287.43  5086.2 2285.81  5267.5 2287.09  5314.6 2288.55  5390.8 2293.68
  5496.0 2303.45  5595.7 2315.14  5637.4 2320.75  5724.4 2335.23  5757.1 2337.64
#Mann=3,-1,0
  3898.9    0.05       0  4996.6    0.05       0  5012.6    0.05       0
Bank Sta=4996.6,5012.6
Exp/Cntr=0.3,0.1

Type RM Length L Ch R = 1,102390,552,552,552
BEGIN DESCRIPTION:
Buffalo Creek 123.0
END DESCRIPTION:
XS GIS Cut Line= 3
      1297605.00      6919188.00      1298405.00      6918388.00
      1298916.65      6917773.36
#Sta/Elev= 30
  3872.3 2312.27  3928.9 2307.42  3957.1 2308.11  4197.6 2294.64  4537.0 2284.67
  4692.5 2282.87  4805.7 2284.84  4834.0 2276.95  4848.1 2276.03  4933.0 2275.58
  4975.4 2278.45  4992.1 2273.04  4993.6 2272.54  5008.1 2273.04  5060.3 2276.60
  5068.1 2279.24  5074.6 2277.97  5081.7 2280.59  5109.8 2283.35  5117.6 2287.22
  5124.1 2287.01  5131.9 2290.30  5138.4 2288.26  5146.2 2291.44  5152.7 2289.09
  5159.8 2293.76  5358.4 2299.88  5458.7 2305.38  5586.2 2314.89  5803.4 2335.56
#Mann=3,-1,0
  3872.3    0.05       0  4992.1   0.033       0  5008.1    0.05       0
Bank Sta=4992.1,5008.1
Exp/Cntr=0.3,0.1

Type RM Length L Ch R = 1,101838,532,532,532
BEGIN DESCRIPTION:
Buffalo Creek 122.0
END DESCRIPTION:
XS GIS Cut Line= 3
      1297755.03      6919287.98      1298555.00      6918738.00
      1299255.00      6917938.00
#Sta/Elev= 30
  4024.0 2308.64  4103.1 2303.28  4109.2 2303.91  4168.8 2301.23  4218.1 2300.41
  4303.3 2295.88  4563.2 2288.75  4613.9 2286.20  4649.8 2285.44  4655.8 2283.51
  4670.7 2282.89  4727.8 2282.30  4764.2 2283.28  4837.0 2282.39  4843.9 2283.20
  4900.7 2281.61  4930.5 2276.41  4951.5 2274.39  4998.1 2271.92  5008.1 2269.62
  5009.6 2269.12  5024.1 2269.62  5044.6 2272.51  5058.8 2277.95  5073.1 2285.19
  5165.1 2289.71  5327.4 2294.88  5653.9 2311.50  5788.7 2320.24  6057.8 2341.75
#Mann=3,-1,0
  4024.0    0.05       0  5008.1   0.033       0  5024.1    0.05       0
Bank Sta=5008.1,5024.1
Exp/Cntr=0.3,0.1

Type RM Length L Ch R = 1,101306,557,557,557
BEGIN DESCRIPTION:
Buffalo Creek 121.0
END DESCRIPTION:
XS GIS Cut Line= 3
      1298355.02      6919637.98      1298905.00      6919038.00
      1299454.98      6918238.03
#Sta/Elev= 30
  4186.2 2305.10  4242.6 2302.72  4292.5 2298.08  4313.5 2298.18  4419.6 2291.63
  4504.7 2288.19  4766.7 2283.04  4801.9 2281.79  4851.2 2277.74  4907.9 2281.13
  4993.0 2279.74  5003.1 2278.30  5007.6 2268.32  5020.5 2266.94  5022.0 2266.44
  5036.5 2266.94  5043.4 2272.65  5049.5 2272.44  5058.3 2274.46  5085.3 2275.04
  5151.0 2279.75  5194.3 2285.68  5381.0 2290.65  5575.2 2299.39  5769.3 2311.94
  5898.1 2322.69  5921.6 2322.36  5927.6 2324.78  5934.5 2325.56  5970.9 2327.85
#Mann=3,-1,0
  4186.2    0.05       0  5020.5    0.05       0  5036.5    0.05       0
Bank Sta=5020.5,5036.5
Exp/Cntr=0.3,0.1

Type RM Length L Ch R = 1,100749,539,539,539
BEGIN DESCRIPTION:
Buffalo Creek 120.0
END DESCRIPTION:
XS GIS Cut Line= 3
      1298654.98      6920138.03      1299205.00      6919388.00
      1299604.99      6918588.02
#Sta/Elev= 30
  4069.9 2307.51  4091.9 2305.08  4198.5 2300.86  4355.2 2292.11  4384.5 2287.40
  4392.4 2289.70  4484.8 2284.59  4570.5 2282.08  4764.4 2278.34  4800.5 2278.65
  4842.2 2276.98  4921.6 2278.12  4942.5 2279.86  4957.2 2275.41  4971.8 2272.96
  4978.0 2272.65  4992.7 2274.97  5002.8 2274.73  5006.0 2263.17  5007.5 2262.67
  5022.0 2263.17  5022.4 2266.07  5053.1 2273.13  5081.0 2274.51  5134.2 2279.56
  5313.0 2282.56  5536.6 2291.00  5782.6 2303.28  5805.0 2305.75  5894.4 2310.83
#Mann=3,-1,0
  4069.9    0.05       0  5006.0    0.05       0  5022.0    0.05       0
Bank Sta=5006,5022
Exp/Cntr=0.3,0.1

Type RM Length L Ch R = 1,100210,666,666,666
BEGIN DESCRIPTION:
Buffalo Creek 119.0
END DESCRIPTION:
XS GIS Cut Line= 3
      1299085.90      6920403.59      1299405.00      6919838.00
      1299919.25      6918745.58
#Sta/Elev= 30
  4350.8 2297.61  4382.7 2293.83  4544.5 2292.11  4647.0 2288.98  4662.9 2285.53
  4678.7 2284.71  4690.3 2287.05  4713.2 2285.07  4787.1 2283.17  4852.1 2277.03
  4862.3 2277.14  4873.9 2272.42  4883.9 2271.17  4948.9 2267.40  4962.6 2263.01
  4964.1 2262.51  4978.6 2263.01  5003.0 2265.64  5014.4 2273.23  5037.1 2274.66
  5133.8 2274.38  5202.2 2277.75  5344.5 2276.63  5430.1 2277.90  5519.7 2280.09
  5652.3 2287.61  5828.7 2295.32  5879.8 2298.91  6022.0 2298.41  6207.6 2303.09
#Mann=3,-1,0
  4350.8    0.05       0  4962.6    0.05       0  4978.6    0.05       0
Bank Sta=4962.6,4978.6
Exp/Cntr=0.3,0.1

Type RM Length L Ch R = 1,99544,449,449,449
BEGIN DESCRIPTION:
Buffalo Creek 118.0
END DESCRIPTION:
XS GIS Cut Line= 3
      1299645.00      6920417.67      1299891.52      6920146.84
      1300023.46      6919105.18
#Sta/Elev= 30
  4271.7 2287.41  4342.1 2282.63  4377.9 2283.58  4413.0 2280.53  4512.4 2276.17
  4533.3 2273.45  4747.6 2270.50  4784.0 2268.39  4789.0 2269.41  4838.3 2269.27
  4864.1 2265.40  4969.4 2263.28  4991.6 2259.01  4993.1 2258.51  5007.6 2259.01
  5050.0 2260.45  5090.3 2265.93  5140.7 2269.87  5160.9 2273.20  5179.5 2272.97
  5184.5 2275.72  5191.1 2276.68  5221.4 2278.70  5424.8 2284.01  5473.4 2283.76
  5483.5 2281.71  5493.5 2281.61  5513.7 2284.28  5574.2 2286.31  5687.9 2292.72
#Mann=3,-1,0
  4271.7    0.05       0  4991.6    0.05       0  5007.6    0.05       0
Bank Sta=4991.6,5007.6
Exp/Cntr=0.3,0.1

Type RM Length L Ch R = 1,99095,623,623,623
BEGIN DESCRIPTION:
Buffalo Creek 117.0
END DESCRIPTION:
XS GIS Cut Line= 3
      1299505.03      6920587.98      1300205.00      6920038.00
      1300474.78      6919227.40
#Sta/Elev= 30
  4103.0 2302.25  4302.7 2290.91  4323.5 2287.56  4352.4 2287.41  4416.6 2281.24
  4437.4 2281.82  4530.4 2276.79  4573.5 2272.69  4722.9 2268.06  4807.9 2268.25
  4901.0 2265.73  4936.2 2259.58  4942.6 2261.00  4957.1 2256.78  4957.2 2255.49
  4958.7 2254.99  4973.2 2255.49  5130.2 2260.63  5140.8 2263.36  5151.3 2262.61
  5198.9 2266.90  5204.1 2269.24  5262.1 2270.96  5267.4 2272.86  5288.3 2272.65
  5309.4 2275.53  5325.4 2274.41  5330.7 2277.00  5673.5 2283.29  5847.5 2290.16
#Mann=3,-1,0
  4103.0    0.05       0  4957.2   0.033       0  4973.2    0.05       0
Bank Sta=4957.2,4973.2
Exp/Cntr=0.3,0.1

Type RM Length L Ch R = 1,98472,482,482,482
BEGIN DESCRIPTION:
Buffalo Creek 116.0
END DESCRIPTION:
XS GIS Cut Line= 3
      1299676.20      6920763.84      1300346.46      6920532.07
      1301095.49      6920425.30
#Sta/Elev= 30
  4290.8 2297.37  4418.8 2293.16  4475.8 2292.71  4564.1 2288.94  4595.2 2286.80
  4600.5 2284.67  4626.4 2280.71  4649.3 2279.77  4688.7 2274.47  4776.3 2269.82
  4829.2 2265.12  4892.6 2262.57  4901.6 2259.39  4913.8 2262.87  4938.1 2261.92
  4956.1 2256.83  4961.3 2252.93  4962.8 2252.43  4977.3 2252.93  5038.9 2259.06
  5049.0 2258.30  5079.3 2263.24  5129.8 2267.46  5135.0 2269.35  5205.8 2274.19
  5271.3 2281.44  5301.6 2286.63  5331.9 2288.82  5453.1 2295.58  5756.6 2302.62
#Mann=3,-1,0
  4290.8    0.05       0  4961.3    0.05       0  4977.3    0.05       0
Bank Sta=4961.3,4977.3
Exp/Cntr=0.3,0.1

Type RM Length L Ch R = 1,97990,547,547,547
BEGIN DESCRIPTION:
Buffalo Creek 115.0
END DESCRIPTION:
XS GIS Cut Line= 3
      1299832.40      6921206.56      1300555.00      6920938.00
      1300955.00      6920838.00
#Sta/Elev= 30
  4218.0 2293.34  4466.1 2280.61  4630.8 2274.58  4686.2 2271.38  4771.9 2268.44
  4857.6 2268.91  4888.0 2263.55  4893.3 2264.07  4913.0 2261.83  4956.9 2260.25
  4979.1 2252.53  4991.5 2251.25  4998.9 2247.31  5000.4 2246.81  5014.9 2247.31
  5019.8 2250.72  5030.1 2254.70  5053.3 2256.02  5081.7 2259.33  5089.4 2262.05
  5112.6 2264.70  5122.9 2268.25  5143.5 2272.96  5184.7 2278.42  5195.0 2282.69
  5213.1 2286.01  5277.5 2288.78  5295.6 2288.22  5336.8 2291.32  5401.2 2293.81
#Mann=3,-1,0
  4218.0    0.05       0  4998.9    0.05       0  5014.9    0.05       0
Bank Sta=4998.9,5014.9
Exp/Cntr=0.3,0.1

Type RM Length L Ch R = 1,97443,534,534,534
BEGIN DESCRIPTION:
Buffalo Creek 114.0
END DESCRIPTION:
XS GIS Cut Line= 3
      1300144.95      6921770.78      1300805.00      6921388.00
      1301471.52      6921098.71
#Sta/Elev= 30
  4232.7 2285.96  4279.0 2286.12  4388.3 2280.50  4548.9 2276.08  4556.4 2277.17
  4741.1 2269.42  4929.0 2257.59  4950.6 2254.86  4960.5 2251.88  4982.1 2249.96
  4984.8 2244.51  4986.3 2244.01  5000.8 2244.51  5017.5 2250.19  5057.1 2254.53
  5086.0 2253.37  5104.0 2255.34  5109.5 2254.24  5156.4 2259.47  5185.3 2260.40
  5208.7 2262.95  5232.2 2262.89  5268.2 2266.92  5284.6 2267.29  5308.0 2265.23
  5322.7 2267.83  5399.1 2268.73  5519.0 2278.08  5658.3 2284.09  5722.3 2288.28
#Mann=3,-1,0
  4232.7    0.05       0  4984.8   0.033       0  5000.8    0.05       0
Bank Sta=4984.8,5000.8
Exp/Cntr=0.3,0.1

Type RM Length L Ch R = 1,96909,589,589,589
BEGIN DESCRIPTION:
Buffalo Creek 113.0
END DESCRIPTION:
XS GIS Cut Line= 3
      1300487.85      6921992.13      1301055.00      6921838.00
      1301775.82      6921532.52
#Sta/Elev= 30
  4408.0 2281.78  4570.9 2275.80  4710.2 2268.68  4840.3 2255.44  4864.2 2254.50
  4881.7 2255.65  4933.4 2251.05  4943.9 2245.52  4977.4 2243.54  4978.9 2243.04
  4993.4 2243.54  5010.3 2244.80  5017.4 2249.12  5039.4 2253.70  5192.3 2253.87
  5310.7 2258.85  5339.8 2262.63  5368.9 2263.45  5392.6 2266.54  5445.3 2269.58
  5521.8 2276.86  5545.5 2280.94  5550.9 2280.60  5569.1 2288.19  5574.6 2284.97
  5669.1 2291.47  5703.8 2297.75  5751.2 2299.50  5756.6 2298.46  5778.6 2300.95
#Mann=3,-1,0
  4408.0    0.05       0  4977.4   0.033       0  4993.4    0.05       0
Bank Sta=4977.4,4993.4
Exp/Cntr=0.3,0.1

Type RM Length L Ch R = 1,96320,533,533,533
BEGIN DESCRIPTION:
Buffalo Creek 112.0
END DESCRIPTION:
XS GIS Cut Line= 4
      1301067.09      6922250.56      1301330.00      6922213.00
      1301505.00      6922188.00      1302059.01      6921887.96
#Sta/Elev= 30
  4557.4 2271.74  4676.5 2273.79  4747.2 2270.98  4757.3 2269.93  4797.7 2258.59
  4823.0 2256.50  4868.4 2258.09  4878.5 2255.50  4918.9 2252.98  4959.4 2243.95
  4971.6 2238.58  4973.1 2238.08  4987.6 2238.58  4989.7 2240.63  5002.6 2241.58
  5045.2 2251.65  5051.6 2249.79  5057.3 2252.34  5073.5 2253.20  5079.4 2251.34
  5111.5 2256.36  5199.0 2263.32  5204.7 2265.64  5215.2 2264.80  5220.9 2267.07
  5237.1 2265.93  5242.8 2268.18  5302.7 2270.09  5412.0 2279.72  5629.8 2291.17
#Mann=3,-1,0
  4557.4    0.05       0  4971.6    0.05       0  4987.6    0.05       0
Bank Sta=4971.6,4987.6
Exp/Cntr=0.3,0.1

Type RM Length L Ch R = 1,95787,525,525,525
BEGIN DESCRIPTION:
Buffalo Creek 111.0
END DESCRIPTION:
XS GIS Cut Line= 3
      1300957.45      6923109.32      1301605.00      6922688.00
      1302030.03      6922412.98
#Sta/Elev= 30
  4223.8 2275.89  4418.2 2270.14  4424.2 2271.53  4650.4 2263.17  4735.2 2258.17
  4771.4 2253.78  4780.6 2255.94  4786.5 2252.70  4807.6 2251.80  4816.8 2253.23
  4822.8 2251.20  4880.1 2246.24  4895.2 2246.75  4901.2 2244.12  4937.4 2239.99
  4988.8 2238.85  4999.3 2236.82  5001.0 2234.90  5002.5 2234.40  5018.7 2234.90
  5040.2 2237.98  5091.6 2240.23  5133.9 2249.85  5139.8 2249.58  5149.0 2252.86
  5206.4 2260.24  5234.6 2267.89  5329.9 2270.60  5357.5 2275.04  5502.6 2282.68
#Mann=3,-1,0
  4223.8    0.05       0  5001.0    0.05       0  5018.7    0.05       0
Bank Sta=5001,5018.7
Exp/Cntr=0.3,0.1

Type RM Length L Ch R = 1,95262,432,432,432
BEGIN DESCRIPTION:
Buffalo Creek 110.0
END DESCRIPTION:
XS GIS Cut Line= 3
      1301637.29      6924087.79      1301955.00      6923038.00
      1302179.99      6922363.03
#Sta/Elev= 30
  3902.7 2296.49  4059.2 2294.66  4227.2 2286.54  4364.1 2277.36  4539.8 2260.97
  4638.0 2257.10  4671.0 2253.20  4676.2 2254.28  4736.8 2247.93  4748.8 2248.32
  4780.2 2242.17  4807.9 2241.33  4813.2 2239.46  4832.4 2242.09  4840.9 2248.48
  4846.1 2240.38  4853.2 2243.52  4895.0 2238.12  4936.8 2238.51  4969.0 2230.24
  4970.5 2229.74  4986.7 2230.24  4989.1 2233.28  5020.6 2235.59  5083.8 2246.88
  5115.5 2250.04  5410.6 2270.36  5547.6 2277.67  5568.7 2280.67  5711.0 2288.40
#Mann=3,-1,0
  3902.7    0.05       0  4969.0    0.05       0  4986.7    0.05       0
Bank Sta=4969,4986.7
Exp/Cntr=0.3,0.1

Type RM Length L Ch R = 1,94830,619,619,619
BEGIN DESCRIPTION:
Buffalo Creek 109.0
END DESCRIPTION:
XS GIS Cut Line= 3
      1301981.02      6924067.01      1302204.02      6923306.57
      1302350.82      6922473.27
#Sta/Elev= 30
  4230.1 2291.48  4312.4 2288.46  4375.0 2281.94  4447.9 2277.62  4885.6 2257.93
  4896.0 2256.30  4901.5 2253.51  4906.7 2255.05  4934.9 2246.20  4940.1 2241.18
  4948.1 2237.68  4958.5 2234.60  4973.5 2233.70  4991.4 2228.42  4992.9 2227.92
  5009.1 2228.42  5012.1 2231.33  5031.3 2234.09  5102.3 2234.61  5143.0 2238.13
  5214.0 2238.61  5234.7 2243.42  5254.7 2243.21  5283.8 2247.88  5315.6 2248.83
  5386.7 2255.02  5407.5 2259.23  5528.8 2264.27  5660.8 2276.62  5868.7 2286.85
#Mann=3,-1,0
  4230.1    0.05       0  4991.4    0.05       0  5009.1    0.05       0
Bank Sta=4991.4,5009.1
Exp/Cntr=0.3,0.1

Type RM Length L Ch R = 1,94211,564,564,564
BEGIN DESCRIPTION:
Buffalo Creek 108.0
END DESCRIPTION:
XS GIS Cut Line= 3
      1302126.85      6924494.09      1302705.00      6923438.00
      1303147.70      6922613.86
#Sta/Elev= 30
  3796.0 2288.37  4175.4 2274.12  4373.0 2264.68  4485.5 2262.92  4654.3 2256.84
  4801.3 2246.67  4823.1 2241.71  4839.2 2243.40  4844.9 2241.75  4874.6 2241.38
  4910.4 2236.33  4926.5 2237.55  4932.2 2234.86  4977.2 2234.89  4991.9 2230.46
  4999.2 2224.02  5000.7 2223.52  5017.0 2224.02  5030.0 2232.42  5045.4 2235.13
  5102.1 2238.83  5161.5 2245.05  5177.8 2248.85  5205.4 2251.78  5295.1 2258.72
  5533.3 2270.91  5703.0 2282.14  5812.6 2285.33  5872.7 2290.40  5935.5 2290.95
#Mann=3,-1,0
  3796.0    0.05       0  4999.2    0.05       0  5017.0    0.05       0
Bank Sta=4999.2,5017
Exp/Cntr=0.3,0.1

Type RM Length L Ch R = 1,93647,581,581,581
BEGIN DESCRIPTION:
Buffalo Creek 107.0
END DESCRIPTION:
XS GIS Cut Line= 3
      1302923.74      6924598.25      1303105.00      6923838.00
      1303267.46      6922832.80
#Sta/Elev= 30
  4214.0 2284.10  4366.8 2275.42  4389.0 2275.10  4456.2 2270.86  4714.1 2258.09
  4810.5 2254.94  4882.5 2254.57  4887.7 2250.12  4903.0 2246.60  4923.6 2244.18
  4985.3 2233.37  5005.7 2230.96  5015.0 2221.73  5016.5 2221.23  5032.8 2221.73
  5036.1 2225.66  5046.2 2229.97  5056.3 2232.43  5090.7 2233.33  5096.9 2234.96
  5127.2 2238.95  5238.7 2240.05  5280.9 2241.78  5471.7 2253.12  5713.0 2265.47
  5856.6 2275.07  5897.1 2275.84  5947.8 2279.31  5970.1 2278.87  6013.8 2279.97
#Mann=3,-1,0
  4214.0    0.05       0  5015.0    0.05       0  5032.8    0.05       0
Bank Sta=5015,5032.8
Exp/Cntr=0.3,0.1

Type RM Length L Ch R = 1,93066,547,547,547
BEGIN DESCRIPTION:
Buffalo Creek 106.0
END DESCRIPTION:
XS GIS Cut Line= 3
      1303376.87      6924598.21      1303655.00      6923838.00
      1303954.50      6922891.44
#Sta/Elev= 30
  4190.5 2270.75  4695.4 2247.33  4720.6 2244.29  4726.0 2245.25  4733.8 2243.29
  4837.4 2239.99  4861.6 2236.16  4873.3 2236.95  4893.2 2234.19  4898.5 2236.94
  4914.8 2230.26  4959.5 2228.82  4968.0 2224.26  4969.8 2219.66  4971.3 2219.16
  4987.6 2219.66  4990.0 2225.35  4997.3 2229.91  5010.5 2231.71  5031.5 2231.13
  5073.4 2236.38  5182.9 2237.47  5293.7 2248.49  5356.6 2246.87  5511.2 2249.57
  5587.4 2253.79  5671.3 2256.57  5683.3 2258.23  5839.1 2263.43  5992.8 2271.46
#Mann=3,-1,0
  4190.5    0.05       0  4969.8    0.05       0  4987.6    0.05       0
Bank Sta=4969.8,4987.6
Exp/Cntr=0.3,0.1

Type RM Length L Ch R = 1,92519,539,539,539
BEGIN DESCRIPTION:
Buffalo Creek 105.0
END DESCRIPTION:
XS GIS Cut Line= 3
      1303871.67      6924775.28      1304155.00      6923938.00
      1304303.92      6923082.79
#Sta/Elev= 30
  4120.2 2274.65  4176.4 2273.77  4302.1 2265.44  4539.6 2257.34  4655.7 2250.56
  4674.1 2251.64  4679.3 2249.42  4705.5 2251.62  4710.8 2249.56  4729.6 2250.57
  4750.8 2238.34  4773.6 2230.10  4856.3 2228.49  4940.8 2230.31  4957.0 2227.19
  4962.3 2221.87  4963.6 2217.74  4965.1 2217.24  4981.4 2217.74  4993.7 2225.27
  5044.7 2231.80  5091.0 2230.74  5096.1 2233.86  5125.9 2236.56  5227.4 2242.94
  5481.2 2252.16  5531.9 2255.40  5557.6 2259.78  5775.6 2267.71  5872.2 2273.89
#Mann=3,-1,0
  4120.2    0.05       0  4963.6    0.05       0  4981.4    0.05       0
Bank Sta=4963.6,4981.4
Exp/Cntr=0.3,0.1

Type RM Length L Ch R = 1,91980,586,586,586
BEGIN DESCRIPTION:
Buffalo Creek 104.0
END DESCRIPTION:
XS GIS Cut Line= 3
      1304460.21      6924837.77      1304555.00      6924138.00
      1304475.83      6923238.84
#Sta/Elev= 30
  4298.8 2269.01  4429.8 2265.11  4480.2 2261.79  4510.5 2258.60  4518.1 2256.19
  4523.2 2256.99  4540.8 2252.06  4550.8 2250.71  4702.2 2242.53  4722.4 2239.22
  4782.9 2234.30  4833.4 2231.63  4896.1 2230.76  4963.6 2226.55  4968.7 2225.74
  4984.8 2219.80  4993.5 2218.47  4995.0 2217.97  5011.3 2218.47  5015.0 2226.90
  5025.0 2228.65  5055.2 2228.08  5061.1 2230.50  5075.2 2231.40  5225.8 2232.75
  5296.1 2230.88  5376.4 2232.12  5587.2 2247.73  5687.6 2250.20  5907.6 2261.73
#Mann=3,-1,0
  4298.8    0.05       0  4993.5    0.05       0  5011.3    0.05       0
Bank Sta=4993.5,5011.3
Exp/Cntr=0.3,0.1

Type RM Length L Ch R = 1,91394,502,502,502
BEGIN DESCRIPTION:
Buffalo Creek 103.0
END DESCRIPTION:
XS GIS Cut Line= 3
      1304918.53      6924931.60      1305105.00      6924138.00
      1304923.77      6923082.76
#Sta/Elev= 30
  4184.7 2268.04  4332.2 2263.07  4434.9 2257.73  4506.8 2250.60  4541.8 2248.49
  4589.4 2242.14  4631.8 2238.66  4722.6 2233.40  4743.1 2233.81  4759.0 2231.23
  4835.6 2228.43  4897.2 2224.46  4989.6 2226.06  5002.4 2224.74  5010.1 2219.22
  5023.5 2213.12  5025.0 2212.62  5041.3 2213.12  5050.6 2224.68  5070.9 2225.83
  5087.3 2229.05  5092.4 2228.02  5111.5 2231.56  5121.7 2234.91  5182.5 2239.45
  5557.0 2240.31  5742.0 2243.81  5902.9 2250.84  6024.7 2258.29  6070.6 2263.19
#Mann=3,-1,0
  4184.7    0.05       0  5023.5    0.05       0  5041.3    0.05       0
Bank Sta=5023.5,5041.3
Exp/Cntr=0.3,0.1

Type RM Length L Ch R = 1,90892,1009,1009,1009
BEGIN DESCRIPTION:
Buffalo Creek 102.0
END DESCRIPTION:
XS GIS Cut Line= 3
      1305538.33      6924879.49      1305505.00      6924388.00
      1305215.71      6922761.34
#Sta/Elev= 30
  4508.2 2256.94  4589.9 2257.48  4710.2 2260.35  4820.4 2256.88  4920.6 2249.13
  4940.7 2245.91  4950.7 2242.65  4960.7 2237.98  4990.8 2218.74  4998.3 2216.76
  5003.4 2216.76  5011.0 2214.93  5012.2 2213.71  5013.7 2213.21  5030.0 2213.71
  5032.9 2221.39  5041.4 2224.73  5061.8 2225.67  5153.2 2224.63  5253.7 2226.89
  5275.1 2225.97  5305.5 2227.10  5356.3 2226.52  5425.7 2228.56  5489.8 2232.47
  5559.4 2235.04  5955.6 2237.00  6059.8 2238.86  6372.0 2247.85  6653.0 2260.32
#Mann=3,-1,0
  4508.2    0.05       0  5012.2    0.05       0  5030.0    0.05       0
Bank Sta=5012.2,5030
Exp/Cntr=0.3,0.1

Type RM Length L Ch R = 1,89883,810,810,810
BEGIN DESCRIPTION:
Buffalo Creek 101.5
END DESCRIPTION:
XS GIS Cut Line= 4
      1306374.34      6924623.10      1306024.49      6924046.52
      1305675.91      6923434.57      1305699.15      6922807.18
#Sta/Elev= 30
  3901.9 2246.29  3927.5 2240.53  3985.6 2235.81  4043.8 2233.39  4392.7 2230.94
  4620.3 2231.66  4781.7 2223.71  4896.9 2223.36  4954.6 2221.31  4977.4 2221.42
  4986.3 2220.44  4999.0 2209.58  5000.5 2209.08  5016.9 2209.58  5023.4 2210.29
  5029.5 2216.33  5035.3 2220.11  5045.4 2222.01  5081.0 2222.34  5138.5 2231.65
  5153.4 2232.63  5228.4 2234.74  5347.2 2235.95  5447.3 2232.51  5607.4 2235.29
  5827.5 2246.61  5847.5 2248.02  5857.5 2250.34  5887.6 2253.05  5908.4 2256.22
#Mann=3,-1,0
  3901.9    0.05       0  4999.0    0.05       0  5016.9    0.05       0
Bank Sta=4999,5016.9
Exp/Cntr=0.3,0.1

Type RM Length L Ch R = 1,89073,923,923,923
BEGIN DESCRIPTION:
Mapping XS 5ac6d1be
END DESCRIPTION:
XS GIS Cut Line= 3
      1306492.21      6924060.01      1306513.04      6923650.32
      1306100.66      6922721.58
#Sta/Elev= 30
  4308.6 2227.99  4825.1 2225.92  4871.6 2223.80  4907.4 2219.76  4962.1 2217.68
  4970.1 2216.07  4984.5 2208.35  4986.0 2207.85  5002.4 2208.35  5005.8 2217.39
  5022.1 2219.79  5097.4 2221.02  5120.7 2218.96  5137.1 2214.04  5143.9 2218.61
  5149.4 2217.27  5159.0 2219.84  5294.4 2222.75  5476.3 2230.38  5509.1 2234.83
  5531.0 2240.61  5538.0 2246.22  5543.5 2247.05  5584.5 2267.10  5590.0 2266.54
  5613.3 2274.96  5618.7 2273.81  5636.5 2276.61  5659.8 2277.73  5735.0 2279.37
#Mann=3,-1,0
  4308.6    0.05       0  4984.5    0.05       0  5002.4    0.05       0
Bank Sta=4984.5,5002.4
Exp/Cntr=0.3,0.1

Type RM Length L Ch R = 1,88150,381,381,381
BEGIN DESCRIPTION:
Buffalo Creek 100.0
END DESCRIPTION:
XS GIS Cut Line= 5
      1306751.97      6924523.27      1307080.00      6923163.00
      1307055.00      6923038.00      1307024.37      6922941.48
      1306354.98      6922537.99
#Sta/Elev= 30
  3473.3 2228.07  3622.7 2226.03  3977.2 2225.91  4443.3 2222.49  4448.4 2223.22
  4699.8 2217.84  4846.9 2217.25  4918.5 2218.05  4949.1 2216.22  4959.3 2217.06
  4969.4 2214.30  4970.7 2206.72  4972.2 2206.22  4988.6 2206.72  4989.8 2210.45
  4997.5 2212.82  5010.5 2214.21  5016.2 2216.90  5021.4 2217.18  5170.3 2219.08
  5329.5 2224.34  5350.9 2224.22  5366.4 2225.73  5409.1 2226.49  5547.0 2232.19
  5780.0 2244.45  5816.9 2248.95  5853.8 2265.02  5875.1 2268.33  5882.9 2268.08
#Mann=3,-1,0
  3473.3    0.05       0  4970.7    0.05       0  4988.6    0.05       0
Bank Sta=4970.7,4988.6
Exp/Cntr=0.3,0.1

Type RM Length L Ch R = 1,87769,514,514,514
BEGIN DESCRIPTION:
Buffalo Creek 99.5
END DESCRIPTION:
XS GIS Cut Line= 4
      1306980.00      6924263.00      1307430.00      6923013.00
      1307345.63      6922778.23      1306949.15      6922591.64
#Sta/Elev= 30
  3554.9 2224.54  3882.0 2224.34  3974.7 2223.00  4314.8 2221.03  4538.0 2218.74
  4548.6 2217.71  4665.6 2214.86  4673.8 2215.51  4729.3 2214.88  4750.6 2215.86
  4852.7 2216.75  4888.8 2216.08  4899.4 2216.79  4963.1 2214.71  4970.3 2211.83
  4975.4 2206.53  4976.9 2206.03  4993.3 2206.53  5001.0 2215.31  5016.3 2216.00
  5048.1 2214.31  5087.9 2215.49  5170.5 2215.51  5193.3 2216.27  5210.5 2218.63
  5238.9 2220.36  5261.7 2220.88  5409.9 2219.17  5523.4 2220.90  5571.1 2222.61
#Mann=3,-1,0
  3554.9    0.05       0  4975.4    0.05       0  4993.3    0.05       0
Bank Sta=4975.4,4993.3
Exp/Cntr=0.3,0.1
