--- Buffalo Creek Trib 09.prj (project) ---

Proj Title=Buffalo Creek Trib 09 Base Level Engineering
Current Plan=p01
Default Exp/Contr=0.3,0.1
English Units
Geom File=g01
Flow File=f01
Plan File=p01
BEGIN DESCRIPTION:
Buffalo Creek Trib 09
END DESCRIPTION:

--- Buffalo Creek Trib 09.p01 (plan) ---

Plan Title=Multiple Run
Short Identifier=Multiple
Geom File=g01
Flow File=f01
Subcritical Flow
K Sum by GR= 0
Std Step Tol= 0.01
Critical Tol= 0.01
Num of Std Step Trials= 20
Max Error Tol= 0.3
Flow Tol Ratio= 0.001
Split Flow NTrial= 30
Split Flow Tol= 0.02
Split Flow Ratio= 0.02
Log Output Level= 0
Friction Slope Method= 1
Unsteady Friction Slope Method= 2
Unsteady Bridges Friction Slope Method= 1
Parabolic Critical Depth
Global Vel Dist=  1 , 1 , 1
Global Log Level= 0
CheckData=True
Encroach Param= -1, 0, 0, 0
BEGIN DESCRIPTION:
Multiple Run
END DESCRIPTION:

--- Buffalo Creek Trib 09.f01 (steady flow) ---

Flow Title=Multiple
Number of Profiles=7
Profile Names=10-year,25-year,50-year,1pct_min,100-year,1pct_plu,500-year
River Rch & RM= Buffalo Creek Tr,Reach-1,40425
     310     433     534     327     652    1300     985
River Rch & RM= Buffalo Creek Tr,Reach-1,37682
     345     484     598     366     731    1458    1107
River Rch & RM= Buffalo Creek Tr,Reach-1,33647
     501     707     878     539    1076    2147    1639
River Rch & RM= Buffalo Creek Tr,Reach-1,27462
     676     966    1210     749    1495    2984    2316
River Rch & RM= Buffalo Creek Tr,Reach-1,21371
     709    1013    1269     786    1568    3129    2428
River Rch & RM= Buffalo Creek Tr,Reach-1,18538
     774    1113    1399     869    1734    3461    2703
River Rch & RM= Buffalo Creek Tr,Reach-1,14477
     827    1193    1504     937    1870    3731    2930
River Rch & RM= Buffalo Creek Tr,Reach-1,12839
     940    1370    1739    1091    2177    4345    3461
River Rch & RM= Buffalo Creek Tr,Reach-1,10027
    1007    1474    1877    1181    2356    4702    3767
River Rch & RM= Buffalo Creek Tr,Reach-1,8293
    1174    1741    2237    1421    2836    5659    4620
Boundary for River Rch & Prof#=Buffalo Creek Tr,Reach-1,1
Up Type=0
Dn Type=3
Dn Slope=0.005
Boundary for River Rch & Prof#=Buffalo Creek Tr,Reach-1,2
Up Type=0
Dn Type=3
Dn Slope=0.005
Boundary for River Rch & Prof#=Buffalo Creek Tr,Reach-1,3
Up Type=0
Dn Type=3
Dn Slope=0.005
Boundary for River Rch & Prof#=Buffalo Creek Tr,Reach-1,4
Up Type=0
Dn Type=3
Dn Slope=0.005
Boundary for River Rch & Prof#=Buffalo Creek Tr,Reach-1,5
Up Type=0
Dn Type=3
Dn Slope=0.005
Boundary for River Rch & Prof#=Buffalo Creek Tr,Reach-1,6
Up Type=0
Dn Type=3
Dn Slope=0.005
Boundary for River Rch & Prof#=Buffalo Creek Tr,Reach-1,7
Up Type=0
Dn Type=3
Dn Slope=0.005

--- Buffalo Creek Trib 09.g01 (geometry) ---

Geom Title=Existing Conditions

River Reach=Buffalo Creek Tr,Reach-1
Reach XY= 30
      1278805.00      6923088.00      1280984.97      6922438.07
      1283801.95      6923530.24      1284965.22      6923448.30
      1285396.05      6923831.33      1285647.91      6924738.00
      1285255.24      6925853.22      1285452.95      6926682.16
      1284815.95      6926777.63      1284905.00      6927588.00
      1286644.22      6928828.32      1287238.30      6930571.62
      1287908.43      6930445.39      1288904.79      6931080.99
      1289547.54      6930844.09      1290510.09      6928535.70
      1291849.29      6927090.58      1291960.56      6926293.62
      1293549.39      6925282.41      1293662.81      6924681.81
      1295048.95      6922995.46      1295353.50      6923134.53
      1296079.96      6922637.51      1296574.99      6923038.06
      1297939.17      6923037.36      1298260.97      6922690.14
      1299184.96      6922637.39      1300589.80      6922887.50
      1301355.01      6922295.08      1301605.00      6922638.00

Type RM Length L Ch R = 1,40425,449,449,449
BEGIN DESCRIPTION:
Buffalo Creek Trib 09 56.0
END DESCRIPTION:
XS GIS Cut Line= 5
      1278280.00      6925012.99      1279078.04      6923254.80
      1279055.00      6923038.00      1279001.65      6922831.19
      1277980.01      6921613.01
#Sta/Elev= 30
  2846.9 2406.98  3028.1 2405.74  3060.1 2406.94  3105.0 2405.09  3709.0 2402.12
  3752.9 2403.40  3790.9 2401.85  4349.2 2399.67  4378.9 2398.09  4562.4 2396.13
  4591.0 2397.37  4675.4 2394.81  4865.0 2395.03  5011.1 2391.49  5011.4 2390.99
  5015.8 2391.49  5068.0 2394.01  5192.0 2394.62  5223.7 2396.03  5435.8 2396.50
  5486.5 2398.09  5528.2 2397.36  5670.3 2400.34  5996.6 2403.82  6053.8 2406.26
  6096.7 2405.23  6252.8 2408.18  6302.2 2407.59  6686.3 2411.78  6799.2 2412.65
#Mann=4,-1,0
  2846.9   0.045       0  5011.1   0.045       0  5015.8   0.045       0
  6686.3   0.035       0
Bank Sta=5011.1,5015.8
Exp/Cntr=0.3,0.1

Type RM Length L Ch R = 1,39976,449,449,449
BEGIN DESCRIPTION:
Buffalo Creek Trib 09 55.0
END DESCRIPTION:
XS GIS Cut Line= 5
      1278756.22      6925229.41      1279477.34      6923089.87
      1279455.00      6922888.00      1279425.26      6922714.87
      1278755.00      6921988.00
#Sta/Elev= 30
  2539.1 2405.19  3046.9 2402.36  3089.3 2403.35  3272.5 2401.10  3310.9 2402.28
  3367.0 2400.56  3574.8 2400.06  3618.9 2401.22  3681.8 2399.86  3991.4 2399.49
  4482.3 2395.50  4521.3 2396.52  4552.8 2394.90  4756.7 2394.83  4795.2 2393.24
  4939.6 2392.68  4987.5 2390.63  4987.8 2390.13  4992.4 2390.63  5071.0 2392.64
  5131.9 2392.08  5152.5 2393.60  5187.6 2392.77  5280.1 2394.99  5392.9 2395.02
  5421.3 2396.69  5725.8 2398.65  5760.9 2400.37  6114.8 2403.82  6164.4 2405.74
#Mann=3,-1,0
  2539.1   0.045       0  4987.5   0.045       0  4992.4   0.045       0
Bank Sta=4987.5,4992.4
Exp/Cntr=0.3,0.1

Type RM Length L Ch R = 1,39527,862,862,862
BEGIN DESCRIPTION:
Buffalo Creek Trib 09 54.0
END DESCRIPTION:
XS GIS Cut Line= 4
      1279244.50      6924654.33      1279855.00      6922838.00
      1279867.97      6922636.74      1279255.00      6921638.00
#Sta/Elev= 30
  3079.4 2400.51  3212.7 2399.86  3251.6 2401.24  3446.0 2399.39  3477.5 2400.65
  3655.8 2398.38  4331.0 2396.21  4373.1 2397.34  4417.8 2395.71  4606.9 2395.92
  4638.4 2394.26  4963.9 2391.90  4992.9 2389.58  5055.7 2390.04  5074.6 2388.51
  5075.0 2388.01  5079.6 2388.51  5085.8 2390.57  5105.8 2390.96  5242.7 2391.22
  5445.0 2394.90  5475.8 2393.77  5570.6 2396.30  5707.9 2396.43  5924.5 2399.22
  5961.2 2401.11  6034.6 2400.42  6092.6 2402.51  6135.2 2401.48  6369.1 2405.12
#Mann=3,-1,0
  3079.4   0.045       0  5074.6   0.045       0  5079.6   0.045       0
Bank Sta=5074.6,5079.6
Exp/Cntr=0.3,0.1

Type RM Length L Ch R = 1,38665,983,983,983
BEGIN DESCRIPTION:
Buffalo Creek Trib 09 53.5
END DESCRIPTION:
XS GIS Cut Line= 4
      1279533.85      6924639.63      1280652.49      6922731.36
      1280586.69      6922380.42      1280214.31      6921241.38
#Sta/Elev= 30
  2580.5 2400.12  2772.1 2400.46  2809.3 2398.77  3342.9 2396.27  3882.2 2396.22
  4329.8 2393.55  4431.4 2391.16  4460.2 2392.93  4746.1 2388.86  4856.1 2389.72
  4971.4 2387.83  5016.3 2385.31  5016.7 2384.81  5021.4 2385.31  5081.6 2388.87
  5162.6 2388.64  5183.6 2390.91  5215.2 2389.39  5297.0 2390.37  5328.8 2392.77
  5360.7 2391.18  5572.9 2393.18  5615.0 2395.62  5646.6 2394.07  5780.3 2394.75
  6003.4 2398.40  6040.5 2400.83  6099.0 2400.17  6136.1 2402.66  6347.9 2403.21
#Mann=3,-1,0
  2580.5   0.045       0  5016.3   0.045       0  5021.4   0.045       0
Bank Sta=5016.3,5021.4
Exp/Cntr=0.3,0.1

Type RM Length L Ch R = 1,37682,448,448,448
BEGIN DESCRIPTION:
Buffalo Creek Trib 09 53.0
END DESCRIPTION:
XS GIS Cut Line= 4
      1279711.12      6924600.01      1281420.05      6922834.66
      1281505.00      6922638.00      1281425.57      6921031.59
#Sta/Elev= 30
  2323.6 2399.58  3133.9 2394.88  4512.9 2390.58  4562.5 2391.93  4654.4 2389.14
  4718.2 2390.15  4787.9 2386.96  4951.3 2386.25  4988.8 2383.27  4989.3 2382.77
  4995.5 2383.27  5064.9 2386.48  5195.1 2386.78  5235.1 2389.84  5315.2 2389.41
  5355.3 2392.21  5585.5 2392.51  5635.6 2394.73  5765.8 2393.66  5805.8 2396.02
  6036.1 2396.22  6076.1 2398.40  6116.2 2396.86  6156.2 2399.19  6296.4 2399.32
  6336.5 2402.24  6406.6 2400.77  6466.6 2404.45  6556.7 2404.00  6603.2 2406.60
#Mann=3,-1,0
  2323.6   0.045       0  4988.8   0.045       0  4995.5   0.045       0
Bank Sta=4988.8,4995.5
Exp/Cntr=0.3,0.1

Type RM Length L Ch R = 1,37234,449,449,449
BEGIN DESCRIPTION:
Buffalo Creek Trib 09 52.0
END DESCRIPTION:
XS GIS Cut Line= 4
      1279928.08      6924741.12      1281805.47      6923011.74
      1281905.00      6922788.00      1282011.44      6920986.74
#Sta/Elev= 30
  2197.7 2399.25  2728.4 2394.79  3742.3 2392.27  3861.7 2391.67  3880.7 2391.90
  4088.8 2391.31  4455.2 2390.52  4511.9 2387.68  4625.3 2387.75  4709.8 2385.01
  4940.4 2385.70  5001.8 2382.47  5002.3 2381.97  5008.5 2382.47  5080.1 2386.86
  5335.7 2389.88  5375.8 2392.55  5414.9 2391.13  5616.2 2394.70  5754.7 2393.71
  5796.5 2395.92  6016.9 2395.05  6046.9 2396.99  6177.2 2395.89  6217.2 2397.70
  6397.5 2397.35  6434.3 2399.63  6638.0 2399.53  6688.0 2402.48  6799.5 2401.67
#Mann=7,-1,0
  2197.7   0.045       0  3742.3    0.07       0  3861.7   0.035       0
  3880.7    0.07       0  4088.8   0.045       0  5001.8   0.045       0
  5008.5   0.045       0
Bank Sta=5001.8,5008.5
Exp/Cntr=0.3,0.1

Type RM Length L Ch R = 1,36785,431,431,431
BEGIN DESCRIPTION:
Buffalo Creek Trib 09 51.0
END DESCRIPTION:
XS GIS Cut Line= 4
      1280242.80      6924741.08      1282305.00      6922938.00
      1282380.00      6922713.00      1282250.15      6921127.78
#Sta/Elev= 30
  2256.5 2397.10  2515.1 2394.63  3623.8 2390.77  3761.7 2390.33  4330.0 2388.33
  4422.0 2384.81  4591.9 2385.50  4648.9 2383.48  4953.6 2385.12  5013.5 2381.94
  5014.0 2381.44  5020.2 2381.94  5069.6 2385.11  5175.0 2385.03  5206.6 2387.20
  5318.3 2387.70  5354.4 2389.97  5518.9 2390.26  5549.0 2392.55  5589.2 2391.37
  5759.7 2392.71  5789.8 2394.65  5920.3 2393.89  5960.4 2395.81  5990.5 2394.55
  6221.3 2396.68  6361.7 2396.02  6391.8 2397.85  6512.2 2396.61  6823.5 2399.65
#Mann=5,-1,0
  2256.5   0.045       0  3623.8   0.035       0  3761.7   0.045       0
  5013.5   0.045       0  5020.2   0.045       0
Bank Sta=5013.5,5020.2
Exp/Cntr=0.3,0.1

Type RM Length L Ch R = 1,36354,952,952,952
BEGIN DESCRIPTION:
Buffalo Creek Trib 09 50.0
END DESCRIPTION:
XS GIS Cut Line= 4
      1280904.98      6924238.01      1282607.55      6923251.33
      1282705.00      6923038.00      1282846.94      6920498.51
#Sta/Elev= 30
  2798.0 2392.04  3280.3 2389.92  3404.3 2389.44  4021.0 2386.07  4231.2 2382.43
  4901.4 2381.17  4956.4 2383.81  5010.4 2381.26  5060.4 2383.94  5097.2 2380.86
  5097.7 2380.36  5103.9 2380.86  5581.2 2384.42  5626.9 2387.32  5691.4 2386.43
  5771.5 2390.05  5821.6 2388.95  5921.8 2392.81  5951.8 2391.53  6052.0 2394.09
  6202.2 2393.63  6242.3 2396.01  6345.9 2394.93  6372.5 2396.70  6502.7 2395.92
  6582.8 2397.80  7093.6 2400.60  7122.1 2398.91  7220.0 2401.56  7543.8 2403.38
#Mann=7,-1,0
  2798.0   0.045       0  3280.3   0.035       0  3404.3   0.045       0
  5097.2   0.045       0  5103.9   0.045       0  7122.1   0.035       0
  7220.0   0.045       0
Bank Sta=5097.2,5103.9
Exp/Cntr=0.3,0.1

Type RM Length L Ch R = 1,35402,952,952,952
BEGIN DESCRIPTION:
Buffalo Creek Trib 09 49.0
END DESCRIPTION:
XS GIS Cut Line= 4
      1281649.57      6924433.65      1283378.38      6923569.04
      1283505.00      6923388.00      1283830.00      6920863.02
#Sta/Elev= 30
  2841.7 2388.45  2865.0 2387.50  3418.0 2386.16  3446.4 2384.86  3496.7 2385.10
  3742.6 2380.36  4175.4 2379.83  4324.0 2380.13  4379.6 2378.90  4543.3 2378.61
  4566.0 2378.56  5418.1 2378.33  5526.7 2378.27  5909.7 2377.96  5910.2 2377.46
  5916.4 2377.96  6171.9 2378.20  6422.3 2378.69  6719.7 2379.94  6820.5 2382.69
  6881.0 2381.83  6995.0 2382.81  7102.8 2384.23  7193.6 2387.43  7264.1 2385.84
  7308.0 2386.27  7365.0 2388.75  7435.6 2388.30  7506.1 2390.79  7541.4 2390.68
#Mann=10,-1,0
  2841.7   0.045       0  4175.4   0.035       0  4543.3    0.15       0
  4566.0   0.035       0  5418.1    0.15       0  5526.7   0.035       0
  5909.7   0.035       0  5916.4   0.035       0  6171.9    0.15       0
  6422.3   0.045       0
Bank Sta=5909.7,5916.4
Exp/Cntr=0.3,0.1

Type RM Length L Ch R = 1,34450,803,803,803
BEGIN DESCRIPTION:
Buffalo Creek Trib 09 48.5
END DESCRIPTION:
XS GIS Cut Line= 4
      1282034.36      6924266.74      1284180.00      6923613.00
      1284260.65      6923455.19      1284960.28      6918885.89
#Sta/Elev= 30
  2526.0 2386.02  2683.5 2386.25  2710.0 2384.67  2780.9 2384.88  2988.4 2380.91
  3365.1 2379.83  3628.5 2378.83  3740.2 2378.47  5030.6 2377.53  5031.1 2377.03
  5038.3 2377.53  7009.7 2378.04  7423.9 2378.64  7937.9 2381.32  7977.3 2383.13
  8114.2 2384.18  8200.9 2387.01  8332.4 2387.19  8423.5 2389.17  8646.5 2388.41
  8686.5 2389.72  8727.0 2388.44  8893.2 2389.56  8908.3 2389.62  9155.6 2389.52
  9305.7 2390.25  9374.4 2393.18  9500.9 2394.92  9536.3 2397.20  9568.8 2396.58
#Mann=11,-1,0
  2526.0   0.045       0  3365.1   0.035       0  3628.5    0.15       0
  3740.2   0.035       0  5030.6   0.035       0  5038.3   0.035       0
  7009.7    0.15       0  7423.9   0.045       0  8893.2   0.035       0
  8908.3   0.045       0  9155.6   0.035       0
Bank Sta=5030.6,5038.3
Exp/Cntr=0.3,0.1

Type RM Length L Ch R = 1,33647,701,701,701
BEGIN DESCRIPTION:
Buffalo Creek Trib 09 48.0
END DESCRIPTION:
XS GIS Cut Line= 4
      1282104.97      6924288.01      1284824.72      6923765.49
      1285030.00      6922713.00      1286263.53      6918654.53
#Sta/Elev= 30
  1896.1 2386.14  2637.8 2379.68  3065.7 2378.25  4517.7 2377.88  5498.6 2377.59
  5681.3 2377.73  5914.3 2377.32  5914.8 2376.82  5927.4 2377.32  6156.6 2377.81
  6315.2 2377.86  6416.7 2377.80  6828.0 2377.59  7041.3 2378.34  7158.9 2378.15
  7294.0 2377.93  7687.0 2378.26  7953.2 2378.64  8306.7 2379.42  8497.4 2380.35
  8640.3 2381.35  9265.4 2383.41  9313.3 2385.15  9723.4 2387.38  9761.5 2389.62
  9794.4 2387.50  9865.4 2388.06  9903.5 2390.45  9936.3 2388.44  9979.7 2388.84
#Mann=20,-1,0
  1896.1   0.045       0  2637.8   0.035       0  3065.7   0.035       0
  4517.7   0.045       0  5498.6   0.045       0  5681.3   0.045       0
  5914.3   0.045       0  5927.4   0.045       0  6156.6    0.15       0
  6315.2   0.045       0  6416.7   0.035       0  6828.0    0.15       0
  7041.3   0.045       0  7158.9    0.15       0  7294.0   0.045       0
  7687.0    0.15       0  7953.2   0.035       0  8306.7   0.045       0
  8497.4   0.035       0  8640.3   0.045       0
Bank Sta=5914.3,5927.4
Exp/Cntr=0.3,0.1

Type RM Length L Ch R = 1,32946,571,571,571
BEGIN DESCRIPTION:
Buffalo Creek Trib 09 47.0
END DESCRIPTION:
XS GIS Cut Line= 4
      1282404.96      6924438.01      1285142.43      6923963.40
      1285305.00      6923738.00      1287080.00      6920763.00
#Sta/Elev= 30
  1943.4 2384.27  2024.6 2385.25  2090.2 2382.49  2270.8 2381.60  2371.8 2381.31
  2438.3 2379.81  2586.3 2379.03  2820.3 2378.35  2957.7 2378.01  4526.3 2377.61
  4594.0 2377.62  4695.0 2377.63  4807.7 2377.37  4808.2 2376.87  4821.0 2377.37
  5223.3 2377.84  5286.2 2377.79  6690.7 2377.60  6871.8 2377.91  7083.7 2378.08
  7181.5 2378.17  7470.4 2378.45  7587.6 2378.56  7695.1 2378.87  8070.8 2380.59
  8187.5 2382.34  8193.4 2383.53  8214.8 2384.30  8245.9 2383.44  8463.9 2385.42
#Mann=20,-1,0
  1943.4   0.045       0  2270.8   0.035       0  2371.8   0.045       0
  2586.3   0.035       0  2820.3    0.15       0  2957.7   0.035       0
  4526.3   0.045       0  4594.0    0.15       0  4695.0   0.045       0
  4807.7    0.07       0  4821.0    0.15       0  5223.3   0.035       0
  5286.2    0.15       0  6690.7   0.035       0  6871.8   0.035       0
  7083.7   0.035       0  7181.5    0.15       0  7470.4   0.035       0
  7587.6    0.15       0  7695.1   0.045       0
Bank Sta=4807.7,4821
Exp/Cntr=0.3,0.1

Type RM Length L Ch R = 1,32375,469,469,469
BEGIN DESCRIPTION:
Buffalo Creek Trib 09 46.0
END DESCRIPTION:
XS GIS Cut Line= 3
      1282355.02      6924788.00      1285355.00      6924188.00
      1288557.39      6921745.07
#Sta/Elev= 30
  1940.6 2385.60  2209.0 2384.47  2226.2 2384.43  2310.6 2384.21  2412.2 2384.29
  2736.0 2380.82  3097.7 2379.51  3942.9 2377.73  3943.4 2377.23  3956.3 2377.73
  5821.9 2378.42  5882.1 2378.58  5958.3 2378.98  6520.3 2379.79  6570.2 2381.08
  6634.6 2379.93  7019.2 2381.02  7247.8 2379.78  7468.2 2380.96  8054.2 2380.50
  8081.5 2381.73  8218.4 2380.99  8253.8 2382.55  8282.7 2381.47  8345.6 2383.05
  8673.7 2383.97  8717.3 2385.63  8852.4 2385.34  8887.8 2386.89  9027.8 2386.71
#Mann=11,-1,0
  1940.6   0.045       0  2209.0   0.035       0  2226.2   0.045       0
  2310.6   0.035       0  2412.2   0.045       0  3097.7    0.15       0
  3942.9    0.07       0  3956.3    0.15       0  5821.9   0.045       0
  5882.1    0.12       0  5958.3   0.045       0
Bank Sta=3942.9,3956.3
Exp/Cntr=0.3,0.1

Type RM Length L Ch R = 1,31906,433,433,433
BEGIN DESCRIPTION:
Buffalo Creek Trib 09 45.0
END DESCRIPTION:
XS GIS Cut Line= 3
      1282555.04      6924888.00      1285555.00      6924588.00
      1288555.00      6922788.00
#Sta/Elev= 30
  1989.9 2384.88  2049.1 2384.63  2148.9 2384.98  3165.7 2380.23  4023.3 2379.39
  4023.8 2378.89  4036.7 2379.39  4964.6 2380.21  5463.5 2379.55  5755.1 2379.90
  5821.2 2381.51  5879.5 2380.30  6396.5 2380.41  6427.6 2381.75  6476.2 2380.60
  7467.4 2380.88  7525.7 2382.36  7578.2 2381.16  7731.8 2381.70  7768.7 2383.11
  7811.5 2381.89  8023.3 2382.53  8060.2 2384.44  8095.2 2383.21  8262.4 2383.80
  8293.5 2385.44  8328.5 2384.29  8472.8 2386.50  8495.6 2386.16  8503.4 2387.30
#Mann=6,-1,0
  1989.9   0.045       0  2049.1   0.035       0  2148.9   0.045       0
  4023.3   0.045       0  4036.7   0.045       0  8472.8   0.035       0
Bank Sta=4023.3,4036.7
Exp/Cntr=0.3,0.1

Type RM Length L Ch R = 1,31473,434,434,434
BEGIN DESCRIPTION:
Buffalo Creek Trib 09 44.0
END DESCRIPTION:
XS GIS Cut Line= 3
      1282130.04      6925063.00      1285505.00      6924938.00
      1288505.03      6924037.99
#Sta/Elev= 30
  1616.6 2386.20  1931.8 2386.25  1971.8 2385.02  2096.1 2384.88  2195.3 2385.13
  2352.1 2383.74  3612.9 2380.85  3773.0 2382.30  3853.1 2380.58  4473.5 2381.34
  5003.7 2380.34  5004.2 2379.84  5017.1 2380.34  5056.5 2381.43  5108.7 2380.39
  6268.5 2380.70  6329.4 2382.19  6424.2 2381.13  7131.5 2381.47  7175.9 2382.87
  7217.7 2381.87  7378.6 2382.28  7411.7 2384.29  7477.8 2382.95  7787.7 2384.88
  7867.6 2384.86  7892.0 2386.32  7917.2 2385.35  7938.9 2386.38  8126.0 2386.63
#Mann=7,-1,0
  1616.6   0.045       0  2096.1   0.035       0  2195.3   0.045       0
  5003.7   0.045       0  5017.1   0.045       0  7787.7   0.035       0
  7892.0   0.045       0
Bank Sta=5003.7,5017.1
Exp/Cntr=0.3,0.1

Type RM Length L Ch R = 1,31039,779,779,779
BEGIN DESCRIPTION:
Buffalo Creek Trib 09 43.0
END DESCRIPTION:
XS GIS Cut Line= 3
      1282080.02      6925463.00      1285505.00      6925338.00
      1288204.99      6924438.00
#Sta/Elev= 30
  1576.9 2386.46  1832.1 2385.43  1862.1 2386.33  1912.1 2384.83  1995.6 2384.90
  2094.8 2384.84  2126.2 2384.01  2132.3 2384.92  2262.3 2383.65  3132.9 2381.91
  3613.2 2381.18  3653.3 2382.84  3693.3 2381.21  4103.6 2380.98  4123.6 2381.84
  4173.6 2380.96  4944.1 2380.38  4974.1 2381.33  4994.9 2380.38  4995.4 2379.88
  5008.4 2380.38  6111.0 2382.73  6985.9 2382.40  7091.3 2384.46  7207.2 2383.06
  7481.3 2383.98  7576.1 2385.38  7628.9 2384.50  7815.3 2385.27  7850.2 2386.70
#Mann=6,-1,0
  1576.9   0.045       0  1995.6   0.035       0  2094.8   0.045       0
  4994.9   0.045       0  5008.4   0.045       0  7815.3   0.035       0
Bank Sta=4994.9,5008.4
Exp/Cntr=0.3,0.1

Type RM Length L Ch R = 1,30260,1124,1124,1124
BEGIN DESCRIPTION:
Buffalo Creek Trib 09 42.9
END DESCRIPTION:
XS GIS Cut Line= 3
      1283229.74      6925769.24      1285258.66      6925966.64
      1287320.25      6925407.38
#Sta/Elev= 30
  2941.6 2382.85  3790.8 2381.80  3908.1 2381.00  3951.6 2382.69  3981.7 2381.09
  4320.6 2380.94  4373.6 2381.58  4403.7 2380.92  4875.9 2381.08  5114.6 2380.30
  5115.1 2379.80  5128.1 2380.30  5152.4 2381.36  5181.7 2380.35  5564.3 2381.30
  5587.6 2381.78  5604.2 2383.12  5638.8 2381.91  5805.2 2384.24  5973.7 2385.10
  6094.4 2385.47  6126.4 2386.41  6157.5 2385.45  6499.4 2385.65  6613.4 2387.22
  6672.5 2386.23  6677.7 2386.84  6786.8 2386.07  7055.2 2386.16  7116.2 2386.79
#Mann=5,-1,0
  2941.6   0.045       0  5114.6   0.045       0  5128.1   0.045       0
  5973.7   0.035       0  6094.4   0.045       0
Bank Sta=5114.6,5128.1
Exp/Cntr=0.3,0.1

Type RM Length L Ch R = 1,29136,625,625,625
BEGIN DESCRIPTION:
Buffalo Creek Trib 09 42.7
END DESCRIPTION:
XS GIS Cut Line= 5
      1283800.14      6926538.61      1285124.11      6926683.48
      1285383.66      6926820.63      1285722.87      6926718.44
      1287165.35      6926022.24
#Sta/Elev= 30
  3494.0 2383.29  3534.2 2382.17  3539.3 2382.93  3559.2 2383.03  3625.5 2381.63
  3630.5 2382.38  3710.1 2381.20  4004.6 2381.01  4992.3 2380.15  4992.8 2379.65
  5006.0 2380.15  5059.8 2380.54  5167.4 2380.61  5459.1 2381.57  5483.9 2383.27
  5520.5 2382.11  5738.6 2384.34  5760.7 2385.79  5783.4 2384.72  5820.3 2385.99
  5851.2 2385.05  5878.0 2385.28  5986.8 2385.60  6043.1 2387.24  6075.7 2386.14
  6314.4 2386.60  6387.8 2388.18  6442.1 2387.02  6764.1 2387.94  7075.4 2387.76
#Mann=8,-1,0
  3494.0   0.035       0  4004.6   0.045       0  4992.3   0.035       0
  5006.0   0.045       0  5059.8    0.07       0  5167.4   0.045       0
  5738.6   0.035       0  5878.0   0.045       0
Bank Sta=4992.3,5006
Exp/Cntr=0.3,0.1

Type RM Length L Ch R = 1,28511,1049,1049,1049
BEGIN DESCRIPTION:
Buffalo Creek Trib 09 42.6
END DESCRIPTION:
XS GIS Cut Line= 5
      1283753.54      6926526.02      1284779.49      6926829.31
      1284855.00      6926838.00      1285200.42      6926920.67
      1286947.58      6926547.90
#Sta/Elev= 30
  3859.8 2383.45  4131.4 2381.71  4330.6 2380.49  4339.4 2380.65  4344.6 2382.86
  4377.9 2380.60  4383.1 2382.99  4411.2 2380.75  4416.4 2383.05  4474.9 2382.96
  4521.4 2381.18  4619.7 2381.31  4985.1 2380.28  5062.9 2380.15  5086.4 2380.19
  5190.6 2378.87  5191.1 2378.37  5204.3 2378.87  5244.6 2380.39  5491.3 2380.44
  5542.9 2382.34  5636.4 2381.29  5829.8 2381.49  6105.6 2385.17  6132.5 2385.51
  6453.2 2386.49  6502.7 2388.18  6745.9 2387.70  6784.5 2389.30  7147.3 2388.93
#Mann=13,-1,0
  3859.8   0.035       0  4131.4   0.045       0  4474.9   0.035       0
  4619.7   0.045       0  4985.1   0.035       0  5062.9   0.045       0
  5086.4    0.07       0  5190.6   0.035       0  5204.3    0.07       0
  5491.3   0.035       0  5636.4   0.045       0  6105.6   0.035       0
  6132.5   0.045       0
Bank Sta=5190.6,5204.3
Exp/Cntr=0.3,0.1

Type RM Length L Ch R = 1,27462,419,419,419
BEGIN DESCRIPTION:
Buffalo Creek Trib 09 42.0
END DESCRIPTION:
XS GIS Cut Line= 5
      1284255.00      6929937.99      1284921.48      6927893.79
      1285055.00      6927738.00      1285213.15      6927612.54
      1286530.02      6927213.00
#Sta/Elev= 30
  2644.5 2397.11  2954.5 2395.68  3032.5 2393.92  3191.4 2393.91  3264.9 2391.18
  3463.4 2391.02  3500.6 2388.32  3697.3 2388.28  3723.9 2385.95  3864.6 2386.42
  3920.6 2383.97  4032.9 2385.36  4085.5 2382.88  4253.8 2382.18  4295.8 2383.70
  4327.4 2381.68  4548.3 2381.95  4579.8 2380.20  4929.0 2377.76  4949.8 2379.35
  4987.6 2376.92  4988.1 2376.42  5005.4 2376.92  5042.2 2379.34  5705.2 2382.10
  5757.4 2384.09  6025.3 2385.09  6071.0 2387.24  6539.7 2388.95  6577.8 2390.81
#Mann=6,-1,0
  2644.5   0.035       0  2954.5   0.045       0  3032.5   0.035       0
  3264.9   0.045       0  4987.6   0.045       0  5005.4   0.045       0
Bank Sta=4987.6,5005.4
Exp/Cntr=0.3,0.1

Type RM Length L Ch R = 1,27043,465,465,465
BEGIN DESCRIPTION:
Buffalo Creek Trib 09 41.0
END DESCRIPTION:
XS GIS Cut Line= 4
      1284517.96      6930083.95      1285355.00      6927988.00
      1285468.36      6927852.12      1286830.01      6927263.00
#Sta/Elev= 30
  2743.1 2397.65  2900.3 2397.91  3069.7 2394.34  3104.9 2396.00  3147.8 2393.22
  3217.4 2393.02  3263.4 2392.48  3298.7 2393.80  3546.3 2390.74  3600.2 2388.28
  3829.4 2388.22  3869.4 2386.00  4039.6 2386.60  4160.1 2383.96  4201.2 2385.72
  4230.8 2383.17  4440.1 2383.38  4461.6 2381.40  4569.3 2381.97  4637.7 2379.55
  4960.9 2378.68  4988.4 2375.66  4988.9 2375.16  5006.2 2375.66  5260.5 2379.72
  5451.5 2378.83  5632.2 2382.41  5673.8 2381.19  6187.1 2389.27  6660.6 2390.29
#Mann=5,-1,0
  2743.1   0.045       0  3217.4   0.035       0  3263.4   0.045       0
  4988.4   0.045       0  5006.2   0.045       0
Bank Sta=4988.4,5006.2
Exp/Cntr=0.3,0.1

Type RM Length L Ch R = 1,26578,1027,1027,1027
BEGIN DESCRIPTION:
Buffalo Creek Trib 09 40.0
END DESCRIPTION:
XS GIS Cut Line= 4
      1284743.66      6930335.69      1285755.00      6928188.00
      1285843.36      6928018.79      1286979.97      6927463.02
#Sta/Elev= 30
  2626.6 2397.09  2755.0 2397.97  2806.1 2395.45  2948.4 2394.29  2988.4 2396.08
  3022.3 2393.31  3090.6 2392.84  3176.3 2393.63  3220.5 2391.26  3438.0 2390.75
  3506.4 2387.92  3722.5 2388.20  3773.6 2385.75  3933.2 2386.46  3972.5 2384.35
  4194.9 2385.44  4235.0 2383.08  4468.4 2383.22  4624.7 2379.72  4969.1 2377.55
  4988.7 2375.01  4989.2 2374.51  5006.7 2375.01  5045.6 2377.13  5471.5 2378.95
  5573.0 2382.20  5635.0 2381.43  6061.5 2388.55  6096.4 2390.66  6456.6 2390.95
#Mann=5,-1,0
  2626.6   0.045       0  3090.6   0.035       0  3220.5   0.045       0
  4988.7   0.045       0  5006.7   0.045       0
Bank Sta=4988.7,5006.7
Exp/Cntr=0.3,0.1

Type RM Length L Ch R = 1,25551,885,885,885
BEGIN DESCRIPTION:
Buffalo Creek Trib 09 39.3
END DESCRIPTION:
XS GIS Cut Line= 2
      1285138.00      6930836.04      1287123.06      6927545.89
#Sta/Elev= 30
  2437.4 2394.80  2590.4 2392.64  2668.2 2393.72  2734.4 2390.86  2907.0 2390.66
  2949.7 2388.04  3066.2 2387.01  3147.5 2388.25  3213.7 2385.60  3388.4 2386.35
  3446.6 2384.24  3600.0 2383.85  3642.7 2385.67  3722.3 2383.22  3970.7 2384.36
  4013.4 2382.63  4225.0 2383.66  4261.9 2381.49  4502.3 2381.93  4890.1 2374.77
  4982.7 2372.64  4983.2 2372.14  5000.8 2372.64  5007.3 2373.06  5095.4 2377.80
  5208.0 2378.51  5310.1 2378.96  5378.0 2381.96  5857.1 2391.72  6280.0 2391.77
#Mann=9,-1,0
  2437.4   0.045       0  2590.4   0.035       0  2734.4   0.045       0
  4890.1    0.07       0  4982.7   0.045       0  5000.8    0.07       0
  5007.3   0.035       0  5095.4    0.07       0  5208.0   0.045       0
Bank Sta=4982.7,5000.8
Exp/Cntr=0.3,0.1

Type RM Length L Ch R = 1,24666,211,211,211
BEGIN DESCRIPTION:
Buffalo Creek Trib 09 39.2
END DESCRIPTION:
XS GIS Cut Line= 3
      1284885.79      6931987.54      1286870.81      6929465.13
      1287111.94      6928062.21
#Sta/Elev= 30
  1694.3 2405.03  2021.4 2398.55  2063.0 2399.70  2127.1 2396.70  2177.3 2397.89
  2220.2 2395.18  2327.7 2395.51  2361.9 2393.27  2462.3 2393.59  2520.4 2391.04
  3031.6 2387.11  3089.4 2388.42  3224.1 2385.36  3267.4 2387.00  3296.3 2384.65
  3437.4 2385.53  3480.7 2383.25  4499.1 2380.13  4712.3 2377.19  4762.9 2374.25
  4898.4 2373.25  4973.3 2370.26  4973.8 2369.76  4991.5 2370.26  5371.5 2376.76
  5519.3 2379.52  5597.7 2380.22  5924.4 2385.84  6196.5 2391.57  6327.6 2391.95
#Mann=10,-1,0
  1694.3   0.045       0  2361.9   0.035       0  2520.4   0.045       0
  4762.9    0.07       0  4973.3    0.07       0  4991.5    0.07       0
  5371.5   0.035       0  5519.3    0.07       0  5597.7   0.035       0
  5924.4   0.045       0
Bank Sta=4973.3,4991.5
Exp/Cntr=0.3,0.1

Type RM Length L Ch R = 1,24455,250,250,250
BEGIN DESCRIPTION:
Buffalo Creek Trib 09 39.4
END DESCRIPTION:
XS GIS Cut Line= 5
      1285431.61      6932354.14      1286812.72      6930613.00
      1286953.81      6929639.67      1287060.14      6929433.51
      1287283.14      6928398.73
#Sta/Elev= 30
  1642.8 2399.98  1816.6 2396.61  1976.5 2395.50  2125.1 2390.62  2183.8 2391.62
  2262.3 2387.70  2312.0 2389.38  2368.1 2385.86  2440.2 2386.67  2496.2 2383.33
  2787.9 2384.46  2880.8 2381.42  2973.8 2382.22  3009.0 2379.41  3101.9 2379.49
  3180.5 2376.20  3244.6 2377.36  3286.2 2374.43  3685.4 2369.60  3871.2 2368.39
  3871.7 2367.89  3889.4 2368.39  4444.9 2373.57  4654.1 2374.66  4759.4 2372.30
  4963.1 2372.43  5008.1 2369.98  5075.2 2373.34  5179.2 2372.86  6139.2 2389.93
#Mann=9,-1,0
  1642.8   0.035       0  1816.6   0.045       0  1976.5   0.035       0
  2125.1   0.045       0  3685.4   0.035       0  3871.2   0.035       0
  3889.4   0.035       0  4444.9   0.045       0  4654.1   0.035       0
Bank Sta=3871.2,3889.4
Exp/Cntr=0.3,0.1

Type RM Length L Ch R = 1,24205,935,935,935
BEGIN DESCRIPTION:
Buffalo Creek Trib 09 39.1
END DESCRIPTION:
XS GIS Cut Line= 5
      1285587.41      6932417.56      1286845.16      6930613.00
      1287060.14      6929754.69      1287102.90      6929588.89
      1287307.60      6928411.12
#Sta/Elev= 30
  1864.7 2399.44  1893.6 2397.59  1985.8 2397.93  2078.5 2394.57  2343.5 2391.53
  2400.5 2387.91  2437.1 2389.45  2473.6 2386.31  2552.1 2386.84  2581.7 2383.75
  2775.4 2381.73  2817.3 2379.02  2912.4 2381.99  3040.7 2382.01  3234.4 2376.58
  3335.6 2377.27  3392.3 2374.33  3808.7 2369.55  4173.8 2367.42  4174.3 2366.92
  4192.0 2367.42  4334.4 2368.20  4352.5 2368.29  4702.5 2371.63  5007.7 2370.99
  5112.5 2373.82  5141.6 2371.54  5317.7 2372.91  5460.8 2375.40  6315.8 2389.92
#Mann=10,-1,0
  1864.7   0.045       0  1893.6   0.035       0  2078.5   0.045       0
  3808.7   0.035       0  4173.8   0.035       0  4192.0   0.035       0
  4334.4    0.07       0  4352.5   0.035       0  5317.7    0.07       0
  5460.8   0.035       0
Bank Sta=4173.8,4192
Exp/Cntr=0.3,0.1

Type RM Length L Ch R = 1,23270,793,793,793
BEGIN DESCRIPTION:
Buffalo Creek Trib 09 39 0.1
END DESCRIPTION:
XS GIS Cut Line= 3
      1285817.98      6932481.06      1287342.40      6930331.53
      1287275.14      6928678.20
#Sta/Elev= 30
  2612.0 2396.26  2663.4 2395.67  2735.8 2395.56  3064.1 2391.05  3171.1 2387.47
  3221.6 2388.81  3328.6 2385.14  3364.3 2386.61  3400.4 2383.83  3479.9 2384.00
  3652.2 2377.55  3756.1 2376.83  3818.5 2375.90  3845.3 2377.25  3881.0 2374.03
  3934.6 2373.77  4113.1 2371.40  4425.9 2366.83  5237.2 2365.59  5237.7 2365.09
  5255.4 2365.59  5314.3 2366.44  5674.6 2370.36  5751.4 2370.31  6122.1 2372.04
  6205.2 2373.91  6388.1 2377.91  6508.3 2379.99  6802.6 2384.45  6901.9 2384.91
#Mann=18,-1,0
  2612.0   0.045       0  2663.4   0.035       0  2735.8   0.045       0
  3756.1   0.035       0  3818.5   0.045       0  3934.6   0.035       0
  4113.1    0.07       0  4425.9   0.035       0  5237.2   0.035       0
  5255.4   0.035       0  5314.3    0.07       0  5674.6   0.035       0
  5751.4    0.07       0  6122.1   0.035       0  6205.2    0.07       0
  6388.1   0.035       0  6508.3    0.07       0  6802.6   0.035       0
Bank Sta=5237.2,5255.4
Exp/Cntr=0.3,0.1

Type RM Length L Ch R = 1,22477,1106,1106,1106
BEGIN DESCRIPTION:
Buffalo Creek Trib 09 39.0
END DESCRIPTION:
XS GIS Cut Line= 3
      1287130.78      6932688.20      1287855.00      6930538.00
      1287330.00      6928813.01
#Sta/Elev= 30
  2723.6 2392.41  3092.5 2388.04  3192.2 2381.47  3501.9 2371.80  3557.4 2371.66
  3620.7 2366.01  3885.1 2366.29  3911.3 2371.02  3942.8 2373.76  4005.8 2370.53
  4053.4 2365.34  4740.6 2364.47  4741.1 2363.97  4758.9 2364.47  5302.6 2365.05
  5386.8 2365.37  5516.6 2365.95  5692.1 2367.49  5755.5 2365.98  5799.1 2367.91
  5943.3 2367.79  5996.0 2370.85  6016.9 2369.61  6036.3 2371.56  6048.2 2369.98
  6252.9 2375.18  6454.3 2379.84  6491.3 2380.33  6727.7 2383.34  6795.6 2384.43
#Mann=12,-1,0
  2723.6   0.035       0  4740.6   0.035       0  4758.9   0.035       0
  5302.6    0.15       0  5386.8   0.035       0  5516.6    0.15       0
  5799.1   0.035       0  5943.3    0.07       0  6252.9   0.035       0
  6454.3    0.07       0  6491.3   0.035       0  6727.7    0.07       0
Bank Sta=4740.6,4758.9
Exp/Cntr=0.3,0.1

Type RM Length L Ch R = 1,21371,593,593,593
BEGIN DESCRIPTION:
Buffalo Creek Trib 09 38.0
END DESCRIPTION:
XS GIS Cut Line= 3
      1288437.11      6932596.92      1288551.69      6930930.25
      1287380.02      6928813.04
#Sta/Elev= 30
  3336.7 2386.06  3374.8 2383.58  3455.9 2382.58  3496.0 2383.04  3586.2 2380.06
  3866.9 2374.00  4028.5 2368.63  4253.2 2365.21  5572.0 2365.09  5622.1 2364.48
  5622.6 2363.98  5641.0 2364.48  5825.2 2364.95  6412.6 2365.60  6456.1 2367.46
  6493.9 2366.36  6532.0 2367.89  6550.4 2369.09  6587.1 2368.19  6610.0 2370.22
  6618.7 2369.30  6667.9 2371.38  6684.0 2371.59  6690.0 2370.83  6874.6 2375.23
  7044.3 2379.39  7080.2 2379.51  7177.5 2382.96  7389.3 2384.27  7427.1 2385.48
#Mann=8,-1,0
  3336.7   0.045       0  4028.5   0.035       0  5622.1   0.035       0
  5641.0   0.035       0  5825.2    0.15       0  6532.0   0.035       0
  6550.4    0.07       0  6874.6   0.035       0
Bank Sta=5622.1,5641
Exp/Cntr=0.3,0.1

Type RM Length L Ch R = 1,20778,586,586,586
BEGIN DESCRIPTION:
Buffalo Creek Trib 09 37.0
END DESCRIPTION:
XS GIS Cut Line= 3
      1289205.00      6932687.97      1289004.81      6931003.16
      1287560.48      6928794.92
#Sta/Elev= 30
  3295.4 2385.92  3315.5 2385.90  3345.7 2383.85  3406.1 2383.96  3421.9 2383.06
  3527.0 2382.41  3592.2 2380.76  3627.7 2380.88  3939.9 2376.31  4224.3 2369.27
  4453.5 2365.27  5023.2 2364.49  5023.7 2363.99  5042.2 2364.49  5832.6 2364.93
  6706.9 2365.54  6769.3 2367.18  6802.5 2366.73  6845.2 2369.53  6851.2 2368.87
  6896.5 2370.80  6923.5 2370.77  6938.6 2372.43  6953.8 2371.26  6968.9 2372.63
  7113.2 2376.50  7322.8 2380.50  7531.4 2384.61  7538.8 2385.64  7630.7 2385.59
#Mann=7,-1,0
  3295.4   0.045       0  4224.3   0.035       0  5023.2   0.035       0
  5042.2   0.035       0  5832.6    0.15       0  6769.3    0.07       0
  7322.8   0.035       0
Bank Sta=5023.2,5042.2
Exp/Cntr=0.3,0.1

Type RM Length L Ch R = 1,20192,889,889,889
BEGIN DESCRIPTION:
Buffalo Creek Trib 09 36.0
END DESCRIPTION:
XS GIS Cut Line= 3
      1289754.99      6933187.96      1289364.19      6930888.58
      1287473.65      6928525.79
#Sta/Elev= 30
  2666.4 2391.12  2701.3 2390.89  3102.5 2385.22  3133.0 2386.48  3176.1 2383.92
  3527.6 2379.40  4004.7 2375.18  4153.7 2370.90  4439.6 2366.51  4589.5 2365.22
  4996.1 2364.46  4996.6 2363.96  5015.2 2364.46  5820.0 2364.80  6812.9 2365.62
  6883.8 2367.39  6926.6 2366.63  7054.6 2373.05  7211.5 2375.33  7225.9 2377.57
  7240.3 2375.90  7494.7 2381.96  7666.1 2386.81  7759.0 2383.87  7808.6 2386.51
  7843.8 2382.37  7957.9 2383.14  7986.3 2386.50  7994.3 2390.90  8024.8 2390.09
#Mann=10,-1,0
  2666.4   0.035       0  2701.3   0.045       0  4153.7   0.035       0
  4439.6    0.15       0  4589.5   0.035       0  4996.1   0.035       0
  5015.2   0.035       0  5820.0    0.15       0  6883.8    0.07       0
  7494.7   0.035       0
Bank Sta=4996.1,5015.2
Exp/Cntr=0.3,0.1

Type RM Length L Ch R = 1,19303,765,765,765
BEGIN DESCRIPTION:
Buffalo Creek Trib 09 35.0
END DESCRIPTION:
XS GIS Cut Line= 3
      1290705.00      6932888.00      1289608.98      6930346.91
      1287604.98      6928587.99
#Sta/Elev= 30
  2222.8 2386.12  2388.6 2385.18  2429.7 2386.42  2473.3 2384.12  2617.2 2383.66
  3126.7 2376.92  3735.9 2377.04  3851.2 2376.85  4003.1 2371.76  4295.4 2366.90
  4482.6 2364.74  4779.2 2364.69  5471.6 2364.44  5472.1 2363.94  5490.8 2364.44
  5821.3 2364.82  6515.5 2365.52  6632.4 2367.39  6664.5 2366.91  6707.2 2369.82
  6749.9 2369.06  6824.9 2371.88  6862.8 2374.15  6891.3 2373.39  7011.8 2376.15
  7026.0 2377.86  7040.2 2376.55  7153.2 2380.46  7424.6 2385.70  7656.6 2389.30
#Mann=11,-1,0
  2222.8   0.035       0  2388.6   0.045       0  3735.9   0.035       0
  4295.4    0.15       0  4779.2   0.035       0  5471.6   0.035       0
  5490.8   0.035       0  5821.3    0.15       0  6632.4   0.045       0
  6824.9    0.07       0  7424.6   0.035       0
Bank Sta=5471.6,5490.8
Exp/Cntr=0.3,0.1

Type RM Length L Ch R = 1,18538,454,454,454
BEGIN DESCRIPTION:
Buffalo Creek Trib 09 34.0
END DESCRIPTION:
XS GIS Cut Line= 3
      1292854.97      6932287.98      1289855.00      6929888.00
      1287454.98      6928287.99
#Sta/Elev= 30
  1170.4 2387.60  1368.2 2385.63  1374.6 2385.67  1611.4 2382.66  2235.7 2379.36
  2359.6 2378.29  3027.3 2371.53  3973.5 2372.02  4051.8 2372.60  4486.4 2365.54
  4838.5 2364.57  4839.0 2364.07  4857.9 2364.57  5912.4 2365.21  6389.9 2365.73
  6471.3 2367.26  6498.0 2366.97  6555.1 2370.19  6657.3 2369.90  6684.3 2371.75
  6792.5 2372.13  6966.7 2375.25  7017.8 2378.14  7066.5 2377.88  7089.9 2380.40
  7183.3 2382.29  7416.8 2387.97  7533.5 2389.37  7650.2 2390.72  7896.7 2392.52
#Mann=15,-1,0
  1170.4   0.045       0  1368.2    0.07       0  1374.6   0.045       0
  2235.7   0.035       0  2359.6   0.045       0  3973.5   0.035       0
  4838.5   0.035       0  4857.9   0.035       0  5912.4    0.15       0
  6471.3   0.045       0  7066.5   0.035       0  7183.3    0.07       0
  7416.8   0.035       0  7533.5    0.07       0  7650.2   0.045       0
Bank Sta=4838.5,4857.9
Exp/Cntr=0.3,0.1

Type RM Length L Ch R = 1,18084,439,439,439
BEGIN DESCRIPTION:
Buffalo Creek Trib 09 33.0
END DESCRIPTION:
XS GIS Cut Line= 3
      1293105.00      6932288.00      1290105.00      6929588.00
      1287704.97      6928387.98
#Sta/Elev= 30
   958.0 2390.91  1103.5 2389.12  1458.4 2384.56  2310.3 2378.08  2385.5 2377.03
  3021.6 2371.31  3513.4 2370.69  4219.3 2371.32  4682.8 2365.39  5087.8 2364.81
  5088.3 2364.31  5107.2 2364.81  5639.0 2365.06  6184.5 2365.71  6237.9 2367.42
  6344.1 2367.04  6425.2 2370.09  6567.7 2370.04  6595.7 2371.95  6657.2 2370.77
  6707.5 2372.73  6836.0 2372.29  7180.1 2380.28  7190.4 2380.40  7266.5 2384.26
  7289.2 2383.78  7422.3 2387.07  7616.6 2390.21  7654.1 2390.73  7677.4 2390.59
#Mann=18,-1,0
   958.0   0.035       0  1103.5    0.07       0  1458.4   0.045       0
  2310.3   0.035       0  2385.5   0.045       0  3021.6    0.07       0
  3513.4   0.045       0  4219.3   0.035       0  5087.8   0.035       0
  5107.2   0.035       0  5639.0    0.15       0  6184.5   0.045       0
  7180.1   0.035       0  7190.4   0.045       0  7289.2    0.07       0
  7422.3   0.035       0  7616.6    0.07       0  7654.1   0.045       0
Bank Sta=5087.8,5107.2
Exp/Cntr=0.3,0.1

Type RM Length L Ch R = 1,17645,429,429,429
BEGIN DESCRIPTION:
Buffalo Creek Trib 09 32.0
END DESCRIPTION:
XS GIS Cut Line= 3
      1293304.97      6932287.97      1290305.00      6929288.00
      1287904.99      6928288.00
#Sta/Elev= 30
   753.5 2391.77   810.2 2391.38   883.7 2391.35  1074.1 2389.86  1523.5 2383.77
  1567.9 2383.67  2328.8 2377.73  2486.8 2375.11  2970.1 2370.64  3094.9 2370.56
  3108.6 2370.53  3437.7 2370.32  4310.7 2370.91  4446.8 2370.09  4582.9 2369.35
  4938.3 2366.30  5072.5 2365.46  5073.0 2364.96  5091.9 2365.46  5596.7 2366.20
  5660.7 2367.53  5906.1 2367.16  6003.6 2369.79  6151.5 2369.31  6274.4 2371.95
  6902.2 2372.51  7090.7 2375.47  7281.9 2383.13  7430.1 2386.49  7596.1 2389.46
#Mann=20,-1,0
   753.5   0.035       0   810.2   0.045       0   883.7   0.035       0
  1074.1   0.045       0  1523.5    0.07       0  1567.9   0.045       0
  2328.8   0.035       0  2486.8   0.045       0  2970.1    0.07       0
  3094.9   0.045       0  3108.6    0.07       0  3437.7   0.045       0
  4310.7   0.035       0  4446.8   0.045       0  4582.9   0.035       0
  4938.3    0.15       0  5072.5    0.07       0  5091.9    0.15       0
  5596.7   0.045       0  7430.1   0.035       0
Bank Sta=5072.5,5091.9
Exp/Cntr=0.3,0.1

Type RM Length L Ch R = 1,17216,416,416,416
BEGIN DESCRIPTION:
Buffalo Creek Trib 09 31.0
END DESCRIPTION:
XS GIS Cut Line= 3
      1293154.98      6931937.98      1290455.00      6928938.00
      1288054.96      6927937.99
#Sta/Elev= 30
   968.8 2390.76  1017.6 2388.99  1264.2 2385.62  1403.4 2383.97  1989.6 2378.95
  2162.5 2377.24  2293.4 2377.08  2434.8 2376.14  2462.5 2373.96  2522.3 2373.41
  2590.3 2371.64  2764.5 2371.26  2984.2 2370.23  3151.5 2370.27  4628.6 2370.38
  4915.3 2369.52  5139.8 2368.40  5140.3 2367.90  5159.2 2368.40  5784.9 2370.29
  5806.5 2371.55  5914.9 2370.52  5982.6 2372.24  6012.4 2370.94  6579.5 2371.19
  6603.3 2372.66  6892.6 2373.14  7099.5 2376.18  7359.5 2385.00  7604.9 2389.95
#Mann=15,-1,0
   968.8   0.035       0  1017.6   0.045       0  1264.2    0.07       0
  1403.4   0.045       0  1989.6   0.035       0  2162.5   0.045       0
  2293.4   0.035       0  2522.3   0.045       0  2764.5    0.07       0
  2984.2   0.035       0  3151.5   0.045       0  4628.6   0.035       0
  4915.3   0.045       0  5139.8   0.045       0  5159.2   0.045       0
Bank Sta=5139.8,5159.2
Exp/Cntr=0.3,0.1

Type RM Length L Ch R = 1,16800,617,617,617
BEGIN DESCRIPTION:
Buffalo Creek Trib 09 30.0
END DESCRIPTION:
XS GIS Cut Line= 3
      1293505.02      6930988.02      1290505.00      6928588.00
      1288161.28      6927559.40
#Sta/Elev= 30
  1169.0 2386.98  1240.3 2384.68  1453.2 2383.97  1513.3 2382.33  1624.4 2381.33
  2200.7 2377.82  2300.0 2375.89  2328.8 2377.31  2364.0 2374.99  2628.7 2373.61
  2752.6 2371.37  4456.2 2369.78  4735.5 2367.51  4859.4 2368.04  4973.2 2366.88
  4973.7 2366.38  4992.6 2366.88  5548.7 2368.55  5589.7 2370.03  5633.4 2368.87
  5874.2 2369.85  5915.5 2371.62  5950.1 2370.35  6090.0 2372.21  6135.7 2370.89
  6659.9 2372.57  6878.3 2376.33  6932.9 2375.86  7227.8 2383.29  7570.4 2389.02
#Mann=9,-1,0
  1169.0   0.045       0  1513.3   0.035       0  1624.4   0.045       0
  2628.7   0.035       0  2752.6   0.045       0  4735.5   0.035       0
  4859.4   0.045       0  4973.2   0.045       0  4992.6   0.045       0
Bank Sta=4973.2,4992.6
Exp/Cntr=0.3,0.1

Type RM Length L Ch R = 1,16183,199,199,199
BEGIN DESCRIPTION:
Buffalo Creek Trib 09 29.0
END DESCRIPTION:
XS GIS Cut Line= 5
      1293805.02      6931038.02      1291430.00      6928313.00
      1290829.89      6928163.11      1290544.26      6928077.26
      1289005.00      6926538.00
#Sta/Elev= 30
   766.7 2391.55  1184.9 2387.16  1227.7 2385.03  1470.1 2383.87  1615.9 2381.69
  2170.4 2375.79  2198.9 2377.18  2240.6 2374.72  2403.9 2374.53  2453.3 2372.42
  2782.7 2372.03  2793.6 2372.72  2829.2 2370.54  2926.7 2370.21  3344.4 2370.11
  3949.5 2369.97  4448.5 2365.84  4868.0 2365.21  4964.4 2365.03  4964.9 2364.53
  4983.9 2365.03  5078.2 2367.16  5198.2 2366.15  5266.1 2366.29  5418.3 2367.78
  5495.2 2366.06  5706.6 2367.75  5712.1 2367.77  6768.0 2373.46  7475.1 2385.85
#Mann=15,-1,0
   766.7   0.045       0  1470.1   0.035       0  1615.9   0.045       0
  2782.7   0.035       0  2793.6   0.045       0  2926.7    0.07       0
  3344.4   0.045       0  4868.0   0.035       0  4964.4   0.035       0
  4983.9   0.035       0  5198.2   0.045       0  5266.1   0.035       0
  5418.3   0.045       0  5706.6   0.035       0  5712.1   0.045       0
Bank Sta=4964.4,4983.9
Exp/Cntr=0.3,0.1

Type RM Length L Ch R = 1,15984,524,524,524
BEGIN DESCRIPTION:
Buffalo Creek Trib 09 28.0
END DESCRIPTION:
XS GIS Cut Line= 5
      1293955.03      6930938.03      1291576.44      6928135.36
      1291034.54      6928017.54      1290461.85      6927871.47
      1289155.02      6926138.02
#Sta/Elev= 30
   597.3 2391.79  1530.7 2382.10  1678.6 2380.28  2066.3 2375.82  2093.9 2377.14
  2122.5 2374.94  2271.9 2374.46  2349.9 2372.14  2714.4 2371.26  3025.1 2370.54
  3197.6 2370.39  4038.3 2367.15  4052.4 2366.95  4059.9 2369.08  4081.0 2365.53
  4123.8 2367.95  4169.8 2366.59  4536.3 2364.44  4613.5 2364.31  4786.4 2365.22
  4827.9 2361.48  4828.4 2360.98  4847.4 2361.48  4849.7 2363.65  4858.3 2364.87
  4878.9 2365.26  5598.0 2366.74  5756.4 2367.37  6583.2 2371.38  7589.7 2388.59
#Mann=14,-1,0
   597.3   0.045       0  1530.7   0.035       0  1678.6   0.045       0
  2714.4   0.035       0  3025.1    0.07       0  3197.6   0.045       0
  4038.3   0.035       0  4169.8   0.045       0  4536.3   0.035       0
  4613.5   0.045       0  4827.9   0.045       0  4847.4   0.045       0
  5598.0   0.035       0  5756.4   0.045       0
Bank Sta=4827.9,4847.4
Exp/Cntr=0.3,0.1

Type RM Length L Ch R = 1,15460,444,444,444
BEGIN DESCRIPTION:
Buffalo Creek Trib 09 27.0
END DESCRIPTION:
XS GIS Cut Line= 3
      1293605.00      6930088.00      1291205.00      6927688.00
      1289555.02      6925888.03
#Sta/Elev= 30
  1610.9 2383.38  1783.9 2381.73  1903.0 2380.28  2219.0 2375.76  2247.3 2377.16
  2473.6 2372.47  2991.6 2371.32  3067.5 2372.64  3095.8 2370.42  3179.1 2370.35
  3606.5 2369.64  3972.4 2368.71  3995.6 2367.94  4085.8 2367.49  4114.8 2369.57
  4142.3 2366.35  4257.2 2367.98  4411.0 2364.65  4982.7 2361.69  4991.6 2359.19
  4992.1 2358.69  5011.4 2359.19  5033.1 2361.95  5072.8 2360.78  5132.3 2363.24
  5819.0 2364.17  6082.0 2366.90  6197.4 2366.61  6682.5 2371.26  7446.8 2387.44
#Mann=16,-1,0
  1610.9   0.045       0  1783.9   0.035       0  1903.0   0.045       0
  2991.6   0.035       0  3179.1    0.07       0  3606.5   0.045       0
  3972.4   0.035       0  3995.6   0.045       0  4114.8   0.035       0
  4257.2   0.045       0  4982.7    0.07       0  4991.6    0.07       0
  5011.4    0.07       0  5072.8   0.045       0  6082.0   0.035       0
  6197.4   0.045       0
Bank Sta=4991.6,5011.4
Exp/Cntr=0.3,0.1

Type RM Length L Ch R = 1,15016,539,539,539
BEGIN DESCRIPTION:
Buffalo Creek Trib 09 26.0
END DESCRIPTION:
XS GIS Cut Line= 3
      1293855.03      6929738.03      1291455.00      6927338.00
      1289654.99      6925687.99
#Sta/Elev= 30
  1605.8 2382.89  1691.4 2382.07  1816.6 2380.33  2454.4 2372.43  3176.4 2371.15
  3260.5 2372.45  3288.8 2370.17  3345.3 2370.29  3373.6 2372.69  3401.9 2369.29
  3441.3 2371.48  3503.6 2370.41  3515.0 2372.08  3590.4 2370.35  4264.6 2364.95
  4307.0 2362.34  4462.6 2360.07  4773.7 2361.59  5000.5 2359.98  5025.5 2357.82
  5026.0 2357.32  5045.3 2357.82  5056.4 2360.22  5131.3 2359.97  6075.7 2366.09
  6139.9 2364.78  6271.6 2366.73  6557.2 2369.70  6918.0 2379.48  7441.8 2388.99
#Mann=13,-1,0
  1605.8   0.045       0  1691.4   0.035       0  1816.6   0.045       0
  3176.4   0.035       0  3441.3   0.045       0  3503.6    0.07       0
  3590.4   0.045       0  5000.5    0.07       0  5025.5   0.045       0
  5045.3    0.07       0  5131.3   0.045       0  6139.9   0.035       0
  6271.6   0.045       0
Bank Sta=5025.5,5045.3
Exp/Cntr=0.3,0.1

Type RM Length L Ch R = 1,14477,539,539,539
BEGIN DESCRIPTION:
Buffalo Creek Trib 09 25.0
END DESCRIPTION:
XS GIS Cut Line= 3
      1294255.00      6929438.00      1291855.00      6927038.00
      1290330.02      6925713.01
#Sta/Elev= 30
  1611.0 2385.76  1667.6 2386.35  2003.5 2380.98  2005.2 2380.92  2473.7 2375.69
  2502.0 2377.07  2597.4 2374.72  2685.8 2375.85  2724.6 2374.31  2813.1 2375.44
  2897.9 2372.40  3110.1 2370.97  3887.9 2370.64  4368.7 2364.78  4552.6 2364.75
  4807.8 2360.09  4877.8 2359.38  4934.4 2356.11  4991.0 2356.23  5001.9 2354.33
  5002.4 2353.83  5022.5 2354.33  5026.5 2356.13  5127.3 2358.89  5255.3 2360.26
  5614.5 2363.44  6203.0 2364.42  6564.8 2368.79  6694.1 2372.26  7025.3 2379.19
#Mann=12,-1,0
  1611.0   0.045       0  2003.5   0.035       0  2005.2   0.045       0
  2597.4   0.035       0  2724.6   0.045       0  4807.8    0.07       0
  5001.9    0.07       0  5022.5    0.07       0  5127.3   0.035       0
  5255.3   0.045       0  6564.8   0.035       0  6694.1   0.045       0
Bank Sta=5001.9,5022.5
Exp/Cntr=0.3,0.1

Type RM Length L Ch R = 1,13938,550,550,550
BEGIN DESCRIPTION:
Buffalo Creek Trib 09 24.0
END DESCRIPTION:
XS GIS Cut Line= 3
      1294154.98      6928987.97      1291955.00      6926588.00
      1290429.30      6925459.21
#Sta/Elev= 30
  1738.8 2382.01  1790.7 2381.85  2022.1 2379.84  2050.5 2377.36  2120.8 2376.83
  2149.1 2379.22  2225.6 2376.70  2807.7 2371.62  2836.0 2372.95  2878.3 2371.20
  3770.2 2370.83  4732.6 2362.02  4838.8 2360.12  4970.3 2351.42  4970.8 2350.92
  4991.0 2351.42  5051.9 2353.93  5158.4 2352.17  5187.6 2354.81  5243.1 2354.06
  5336.1 2360.10  5473.6 2363.34  5916.1 2366.08  5952.4 2364.74  6095.6 2367.49
  6124.9 2366.24  6387.8 2372.22  6421.4 2371.37  6542.0 2373.56  6892.4 2377.52
#Mann=10,-1,0
  1738.8   0.045       0  1790.7   0.035       0  2225.6   0.045       0
  4732.6    0.07       0  4970.3    0.07       0  4991.0    0.07       0
  5243.1   0.035       0  5336.1   0.045       0  6421.4   0.035       0
  6542.0   0.045       0
Bank Sta=4970.3,4991
Exp/Cntr=0.3,0.1

Type RM Length L Ch R = 1,13388,549,549,549
BEGIN DESCRIPTION:
Buffalo Creek Trib 09 23.0
END DESCRIPTION:
XS GIS Cut Line= 3
      1293680.38      6928026.44      1292105.00      6926188.00
      1290909.79      6925229.75
#Sta/Elev= 30
  2574.0 2373.21  2924.5 2370.78  3740.0 2370.74  4380.5 2365.48  4463.3 2366.53
  4697.1 2363.00  4832.1 2355.75  4924.3 2355.93  4966.6 2352.29  5006.3 2348.05
  5006.8 2347.55  5027.1 2348.05  5109.5 2355.96  5208.0 2360.40  5256.3 2361.35
  5336.8 2364.16  5365.6 2361.46  5395.7 2361.75  5508.8 2363.65  5519.7 2363.68
  5756.1 2367.49  5855.3 2367.02  5884.1 2368.93  5948.1 2367.72  5995.3 2370.09
  6139.9 2371.09  6157.4 2371.00  6289.6 2373.72  6319.6 2372.60  6527.0 2375.04
#Mann=14,-1,0
  2574.0   0.045       0  4380.5   0.035       0  4966.6    0.07       0
  5006.3    0.07       0  5027.1    0.07       0  5208.0   0.035       0
  5256.3    0.07       0  5395.7   0.045       0  5508.8    0.07       0
  5519.7   0.045       0  5995.3   0.035       0  6139.9   0.045       0
  6157.4   0.035       0  6319.6   0.045       0
Bank Sta=5006.3,5027.1
Exp/Cntr=0.3,0.1
