--- UCFB HW Trib 16.prj (project) ---

Proj Title=UCFB HW Trib 16 Base Level Engineering
Current Plan=p01
Default Exp/Contr=0.3,0.1
English Units
Geom File=g01
Flow File=f01
Plan File=p01
BEGIN DESCRIPTION:
UCFB HW Trib 16
END DESCRIPTION:

--- UCFB HW Trib 16.p01 (plan) ---

Plan Title=Multiple Run
Short Identifier=Multiple
Geom File=g01
Flow File=f01
Subcritical Flow
K Sum by GR= 0
Std Step Tol= 0.01
Critical Tol= 0.01
Num of Std Step Trials= 20
Max Error Tol= 0.3
Flow Tol Ratio= 0.001
Split Flow NTrial= 30
Split Flow Tol= 0.02
Split Flow Ratio= 0.02
Log Output Level= 0
Friction Slope Method= 1
Unsteady Friction Slope Method= 2
Unsteady Bridges Friction Slope Method= 1
Parabolic Critical Depth
Global Vel Dist=  1 , 1 , 1
Global Log Level= 0
CheckData=True
Encroach Param= -1, 0, 0, 0
BEGIN DESCRIPTION:
Multiple Run
END DESCRIPTION:

--- UCFB HW Trib 16.f01 (steady flow) ---

Flow Title=Multiple
Number of Profiles=7
Profile Names=10-year,25-year,50-year,1pct_min,100-year,1pct_plu,500-year
River Rch & RM= UCFB HW Trib 16,Reach-1,18409
     461     676     863     547    1092    2179    1775
River Rch & RM= UCFB HW Trib 16,Reach-1,12420
     511     754     966     615    1227    2448    2006
River Rch & RM= UCFB HW Trib 16,Reach-1,8351
     779    1171    1519     978    1952    3894    3266
River Rch & RM= UCFB HW Trib 16,Reach-1,3225
    1066    1623    2124    1378    2749    5485    4670
Boundary for River Rch & Prof#=UCFB HW Trib 16,Reach-1,1
Up Type=0
Dn Type=3
Dn Slope=0.005
Boundary for River Rch & Prof#=UCFB HW Trib 16,Reach-1,2
Up Type=0
Dn Type=3
Dn Slope=0.005
Boundary for River Rch & Prof#=UCFB HW Trib 16,Reach-1,3
Up Type=0
Dn Type=3
Dn Slope=0.005
Boundary for River Rch & Prof#=UCFB HW Trib 16,Reach-1,4
Up Type=0
Dn Type=3
Dn Slope=0.005
Boundary for River Rch & Prof#=UCFB HW Trib 16,Reach-1,5
Up Type=0
Dn Type=3
Dn Slope=0.005
Boundary for River Rch & Prof#=UCFB HW Trib 16,Reach-1,6
Up Type=0
Dn Type=3
Dn Slope=0.005
Boundary for River Rch & Prof#=UCFB HW Trib 16,Reach-1,7
Up Type=0
Dn Type=3
Dn Slope=0.005

--- UCFB HW Trib 16.g01 (geometry) ---

Geom Title=Existing Conditions

River Reach=UCFB HW Trib 16,Reach-1
Reach XY= 30
      1289305.00      6938488.00      1290010.93      6938090.23
      1290285.56      6938167.45      1290310.45      6939190.47
      1290861.21      6939345.80      1291194.05      6939778.00
      1290905.55      6940098.64      1291088.51      6940321.85
      1291501.57      6940289.22      1291312.67      6941044.52
      1291714.71      6941148.75      1292052.70      6941582.17
      1293571.71      6942254.63      1293705.42      6942463.00
      1293557.06      6942982.15      1293795.32      6943227.24
      1294605.00      6943688.00      1295657.71      6943793.40
      1296006.46      6944334.46      1296594.53      6944288.93
      1296856.25      6944634.55      1297761.84      6944695.80
      1297762.80      6945144.21      1298491.64      6945574.68
      1298610.45      6946140.47      1299252.39      6946832.73
      1299306.62      6946449.82      1299451.60      6946345.78
      1299860.89      6946636.04      1300255.00      6946588.00

Type RM Length L Ch R = 1,18409,462,462,462
BEGIN DESCRIPTION:
UCFB HW Trib 16 39.0
END DESCRIPTION:
XS GIS Cut Line= 3
      1289799.24      6938608.83      1289655.00      6938338.00
      1289281.59      6937862.17
#Sta/Elev= 30
  4688.0 2303.64  4779.6 2302.58  4847.6 2300.37  4920.8 2296.74  4942.8 2295.17
  4964.7 2291.73  4972.2 2288.70  4984.7 2287.27  4984.9 2286.77  4988.7 2287.27
  5008.4 2288.00  5033.9 2290.90  5103.1 2294.70  5109.3 2294.64  5116.0 2293.35
  5122.3 2294.02  5130.4 2293.27  5151.2 2296.42  5158.8 2295.79  5165.7 2296.38
  5180.1 2294.33  5186.5 2295.86  5194.6 2295.43  5201.0 2296.63  5215.4 2297.44
  5248.2 2297.95  5347.2 2299.47  5386.7 2300.92  5579.6 2309.56  5599.7 2308.74
#Mann=9,-1,0
  4688.0   0.035       0  4984.7   0.035       0  4988.7   0.035       0
  5033.9    0.07       0  5103.1   0.035       0  5158.8    0.07       0
  5248.2   0.035       0  5347.2    0.07       0  5386.7   0.035       0
Bank Sta=4984.7,4988.7
Exp/Cntr=0.3,0.1

Type RM Length L Ch R = 1,17947,485,485,485
BEGIN DESCRIPTION:
UCFB HW Trib 16 38.0
END DESCRIPTION:
XS GIS Cut Line= 3
      1289853.92      6938525.43      1290005.00      6938088.00
      1290002.35      6937672.10
#Sta/Elev= 30
  4543.0 2302.55  4595.4 2302.25  4646.4 2300.69  4736.7 2297.48  4808.4 2294.80
  4834.3 2292.77  4901.9 2289.84  4921.2 2288.20  4927.8 2286.97  4933.1 2287.38
  4952.9 2285.32  4965.3 2285.18  4982.5 2284.61  4982.8 2284.11  4986.8 2284.61
  4990.2 2285.62  4995.5 2284.80  5003.1 2286.38  5008.3 2286.38  5015.8 2288.97
  5025.8 2290.59  5055.8 2293.00  5075.8 2295.53  5085.8 2295.74  5145.8 2300.42
  5215.8 2307.80  5265.6 2310.07  5305.8 2309.95  5385.8 2312.61  5421.7 2313.08
#Mann=7,-1,0
  4543.0   0.035       0  4646.4    0.07       0  4736.7   0.035       0
  4965.3    0.07       0  4982.5    0.07       0  4986.8    0.07       0
  5265.6   0.035       0
Bank Sta=4982.5,4986.8
Exp/Cntr=0.3,0.1

Type RM Length L Ch R = 1,17462,476,476,476
BEGIN DESCRIPTION:
UCFB HW Trib 16 37.0
END DESCRIPTION:
XS GIS Cut Line= 3
      1289879.95      6938541.09      1290305.00      6938338.00
      1290821.30      6938319.78
#Sta/Elev= 30
  4529.0 2302.22  4566.6 2300.95  4596.8 2300.80  4708.1 2297.28  4767.3 2296.54
  4849.9 2291.81  4856.0 2290.78  4930.7 2286.13  4946.1 2285.40  4963.3 2281.95
  5002.6 2282.36  5017.6 2281.50  5018.0 2281.00  5022.2 2281.00  5022.6 2281.50
  5050.1 2282.23  5100.1 2289.16  5136.6 2292.46  5143.5 2292.36  5170.2 2298.00
  5200.2 2300.99  5220.2 2301.62  5230.2 2300.64  5240.2 2298.68  5260.2 2298.95
  5270.2 2302.37  5300.3 2303.84  5350.3 2303.75  5390.3 2304.65  5516.7 2309.70
#Mann=7,-1,0
  4529.0   0.035       0  4596.8    0.07       0  4708.1   0.035       0
  4930.7    0.07       0  5017.6    0.07       0  5022.6    0.07       0
  5136.6   0.035       0
Bank Sta=5017.6,5022.6
Exp/Cntr=0.3,0.1

Type RM Length L Ch R = 1,16986,49,49,49
BEGIN DESCRIPTION:
UCFB HW Trib 16 36.0
END DESCRIPTION:
XS GIS Cut Line= 5
      1289680.01      6938810.83      1290036.39      6938723.71
      1290357.58      6938798.36      1290520.77      6938826.14
      1290742.54      6938622.41
#Sta/Elev= 30
  4305.9 2306.73  4307.2 2306.73  4474.0 2305.76  4546.0 2304.36  4551.2 2301.79
  4578.7 2299.06  4634.5 2297.93  4661.0 2300.20  4669.5 2298.28  4691.9 2298.06
  4753.2 2293.03  4758.3 2293.89  4800.9 2288.80  4806.1 2290.00  4866.4 2286.13
  4886.2 2283.62  4891.3 2285.04  4974.0 2278.43  4974.4 2277.93  4979.0 2278.43
  5032.8 2282.26  5087.9 2289.80  5162.2 2293.16  5167.7 2296.71  5175.5 2297.96
  5184.0 2299.46  5190.8 2297.89  5369.1 2302.43  5467.4 2303.33  5469.2 2303.67
#Mann=8,-1,0
  4305.9   0.035       0  4307.2    0.07       0  4474.0   0.035       0
  4974.0   0.035       0  4979.0   0.035       0  5175.5    0.07       0
  5369.1   0.035       0  5467.4    0.07       0
Bank Sta=4974,4979
Exp/Cntr=0.3,0.1

Type RM Length L Ch R = 1,16937,426,426,426
BEGIN DESCRIPTION:
UCFB HW Trib 16 35.5
END DESCRIPTION:
XS GIS Cut Line= 4
      1289723.75      6938881.34      1290017.12      6938776.77
      1290520.62      6938881.34      1290770.05      6938680.41
#Sta/Elev= 30
  4343.0 2306.78  4484.5 2305.93  4610.6 2303.33  4686.6 2299.96  4744.2 2293.76
  4774.9 2292.06  4836.9 2285.96  4882.0 2283.78  4887.2 2282.27  4897.4 2281.66
  4917.8 2282.32  4948.5 2280.11  4986.8 2272.51  4987.2 2272.01  4991.8 2272.51
  5004.5 2277.07  5020.0 2282.37  5077.3 2288.28  5122.1 2291.10  5132.6 2293.02
  5173.8 2292.63  5210.2 2292.26  5213.2 2294.63  5216.6 2297.31  5231.0 2299.41
  5323.7 2298.44  5373.3 2299.79  5387.7 2298.81  5434.3 2299.42  5489.0 2299.21
#Mann=8,-1,0
  4343.0    0.07       0  4484.5   0.035       0  4986.8   0.035       0
  4991.8   0.035       0  5004.5    0.07       0  5173.8   0.035       0
  5213.2    0.07       0  5434.3   0.035       0
Bank Sta=4986.8,4991.8
Exp/Cntr=0.3,0.1

Type RM Length L Ch R = 1,16511,435,435,435
BEGIN DESCRIPTION:
UCFB HW Trib 16 35.0
END DESCRIPTION:
XS GIS Cut Line= 3
      1290020.55      6939591.85      1290355.00      6939238.00
      1290610.44      6938854.59
#Sta/Elev= 30
  4513.6 2304.23  4605.0 2303.94  4654.0 2304.26  4731.7 2299.33  4766.9 2296.12
  4788.3 2292.28  4802.5 2291.86  4823.5 2287.24  4859.1 2282.23  4887.4 2280.10
  4894.3 2281.03  4965.1 2270.39  4982.7 2270.33  5005.5 2268.55  5005.9 2268.05
  5010.5 2268.55  5023.0 2271.29  5036.5 2276.83  5080.1 2276.09  5144.7 2277.62
  5209.3 2283.15  5230.4 2288.78  5252.8 2291.75  5345.3 2290.53  5397.0 2290.91
  5425.7 2293.50  5446.7 2292.33  5455.8 2297.84  5460.8 2297.50  5461.2 2297.47
#Mann=7,-1,0
  4513.6    0.07       0  4605.0   0.035       0  4982.7    0.07       0
  5005.5    0.07       0  5010.5    0.07       0  5345.3   0.035       0
  5460.8    0.07       0
Bank Sta=5005.5,5010.5
Exp/Cntr=0.3,0.1

Type RM Length L Ch R = 1,16076,473,473,473
BEGIN DESCRIPTION:
UCFB HW Trib 16 34.0
END DESCRIPTION:
XS GIS Cut Line= 4
      1290335.27      6939602.66      1290728.04      6939431.23
      1290755.00      6939338.00      1290855.78      6938911.66
#Sta/Elev= 30
  4474.3 2297.68  4575.6 2294.41  4686.8 2295.08  4709.2 2295.35  4721.5 2295.18
  4726.9 2293.68  4744.9 2295.16  4750.3 2292.88  4768.3 2293.25  4820.6 2288.89
  4849.4 2283.16  4896.3 2278.39  4900.3 2276.94  4958.3 2272.30  4983.1 2271.80
  5002.5 2268.23  5015.9 2263.91  5016.3 2263.41  5021.0 2263.91  5041.0 2264.69
  5060.8 2269.86  5108.2 2274.20  5123.2 2273.05  5150.5 2274.89  5155.6 2273.43
  5192.8 2275.47  5197.9 2274.53  5256.8 2280.66  5389.0 2289.29  5438.0 2291.97
#Mann=7,-1,0
  4474.3   0.035       0  4686.8    0.07       0  4709.2   0.035       0
  4900.3    0.07       0  5015.9    0.07       0  5021.0    0.07       0
  5389.0   0.035       0
Bank Sta=5015.9,5021
Exp/Cntr=0.3,0.1

Type RM Length L Ch R = 1,15603,485,485,485
BEGIN DESCRIPTION:
UCFB HW Trib 16 33.0
END DESCRIPTION:
XS GIS Cut Line= 3
      1290632.54      6939659.10      1291055.00      6939638.00
      1291431.67      6939587.70
#Sta/Elev= 30
  4572.5 2287.66  4652.5 2284.25  4692.4 2281.90  4697.4 2282.13  4705.1 2279.78
  4725.1 2277.54  4735.2 2275.63  4745.2 2274.86  4955.4 2269.50  4965.4 2270.06
  4974.4 2269.42  4985.5 2265.19  4993.0 2260.95  5005.6 2260.49  5013.1 2259.16
  5013.5 2258.66  5017.9 2258.66  5018.3 2259.16  5032.0 2262.22  5037.1 2261.75
  5056.0 2266.22  5066.1 2267.19  5076.2 2267.42  5146.8 2272.98  5167.0 2273.92
  5227.5 2280.41  5256.3 2284.42  5298.1 2287.59  5308.2 2287.65  5375.5 2293.23
#Mann=5,-1,0
  4572.5    0.07       0  4652.5   0.035       0  4974.4    0.07       0
  5013.1    0.07       0  5018.3    0.07       0
Bank Sta=5013.1,5018.3
Exp/Cntr=0.3,0.1

Type RM Length L Ch R = 1,15118,471,471,471
BEGIN DESCRIPTION:
UCFB HW Trib 16 32.0
END DESCRIPTION:
XS GIS Cut Line= 5
      1290670.74      6940100.18      1290954.60      6939955.65
      1291005.00      6939988.00      1291049.65      6940007.73
      1291388.16      6939864.52
#Sta/Elev= 30
  4621.6 2297.23  4671.3 2297.44  4720.0 2287.17  4729.3 2284.72  4761.0 2281.08
  4768.2 2277.75  4773.8 2277.82  4790.4 2273.76  4796.0 2274.46  4812.6 2270.31
  4834.9 2267.40  4895.7 2262.92  4907.2 2265.01  4918.1 2264.37  4923.8 2259.38
  4929.5 2258.42  4937.6 2264.26  4950.2 2266.01  4971.3 2265.52  4977.2 2261.48
  4994.5 2255.04  4994.9 2254.54  4999.7 2255.04  5008.9 2255.98  5014.4 2259.88
  5021.9 2262.19  5043.6 2266.23  5142.5 2266.39  5326.1 2278.79  5416.4 2282.33
#Mann=4,-1,0
  4621.6   0.035       0  4720.0    0.07       0  4994.5    0.07       0
  4999.7    0.07       0
Bank Sta=4994.5,4999.7
Exp/Cntr=0.3,0.1

Type RM Length L Ch R = 1,14647,465,465,465
BEGIN DESCRIPTION:
UCFB HW Trib 16 31.0
END DESCRIPTION:
XS GIS Cut Line= 3
      1290647.41      6940414.42      1291105.00      6940338.00
      1291420.91      6939910.36
#Sta/Elev= 30
  4532.4 2281.80  4658.6 2277.57  4725.4 2277.37  4773.3 2275.02  4786.2 2276.26
  4892.0 2269.04  4925.4 2265.41  4935.5 2262.25  4955.8 2261.22  4976.1 2257.29
  4999.4 2260.53  5003.6 2255.74  5009.9 2256.05  5021.8 2252.88  5022.2 2252.38
  5027.1 2252.88  5032.9 2254.84  5039.1 2254.25  5053.8 2258.45  5068.4 2260.56
  5103.9 2263.08  5133.1 2262.98  5160.2 2260.87  5189.5 2262.85  5224.9 2260.84
  5239.6 2261.46  5375.3 2269.93  5425.4 2275.44  5490.1 2277.55  5528.0 2281.02
#Mann=5,-1,0
  4532.4    0.07       0  4658.6   0.035       0  4892.0    0.07       0
  5021.8    0.07       0  5027.1    0.07       0
Bank Sta=5021.8,5027.1
Exp/Cntr=0.3,0.1

Type RM Length L Ch R = 1,14182,430,430,430
BEGIN DESCRIPTION:
UCFB HW Trib 16 30.0
END DESCRIPTION:
XS GIS Cut Line= 4
      1290794.99      6940532.48      1291434.23      6940330.46
      1291505.00      6940288.00      1291729.98      6940263.00
#Sta/Elev= 30
  4250.8 2273.92  4355.7 2272.91  4446.5 2270.15  4565.4 2268.23  4721.9 2269.02
  4838.1 2263.73  4859.1 2263.76  4890.5 2261.03  4924.6 2260.23  4945.4 2258.01
  4953.2 2255.59  4959.0 2258.23  4968.7 2254.39  4993.3 2251.49  4993.7 2250.99
  4998.6 2251.49  5000.8 2253.41  5013.8 2254.77  5044.0 2264.52  5054.0 2260.24
  5084.2 2264.23  5094.3 2267.52  5114.4 2270.86  5124.5 2273.59  5134.5 2278.41
  5154.7 2285.33  5174.8 2290.36  5191.3 2291.23  5205.0 2291.09  5230.1 2288.72
#Mann=5,-1,0
  4250.8   0.035       0  4721.9    0.07       0  4993.3    0.07       0
  4998.6    0.07       0  5191.3   0.035       0
Bank Sta=4993.3,4998.6
Exp/Cntr=0.3,0.1

Type RM Length L Ch R = 1,13752,449,449,449
BEGIN DESCRIPTION:
UCFB HW Trib 16 29.0
END DESCRIPTION:
XS GIS Cut Line= 3
      1290954.74      6940659.21      1291405.00      6940688.00
      1291761.91      6940673.17
#Sta/Elev= 30
  4548.8 2268.45  4625.0 2266.16  4739.5 2263.03  4749.5 2263.56  4779.5 2261.50
  4819.6 2261.66  4839.7 2262.77  4849.7 2262.24  4869.7 2259.53  4918.2 2256.50
  4949.9 2253.42  4979.9 2252.47  4994.8 2249.53  4995.2 2249.03  5000.1 2249.53
  5010.0 2250.22  5040.0 2255.53  5050.0 2258.11  5080.1 2268.42  5090.1 2270.42
  5110.1 2271.56  5130.1 2275.24  5160.1 2279.03  5190.1 2279.64  5230.2 2281.84
  5250.2 2281.76  5280.2 2279.82  5330.3 2280.63  5350.3 2279.67  5357.2 2278.08
#Mann=4,-1,0
  4548.8   0.035       0  4625.0    0.07       0  4994.8    0.07       0
  5000.1    0.07       0
Bank Sta=4994.8,5000.1
Exp/Cntr=0.3,0.1

Type RM Length L Ch R = 1,13303,433,433,433
BEGIN DESCRIPTION:
UCFB HW Trib 16 28.0
END DESCRIPTION:
XS GIS Cut Line= 5
      1290954.34      6941341.92      1291336.26      6941147.49
      1291355.00      6941088.00      1291371.41      6941031.60
      1291748.55      6940725.64
#Sta/Elev= 30
  4505.4 2272.66  4618.3 2269.55  4696.3 2267.45  4780.2 2262.90  4857.6 2259.14
  4918.8 2259.31  4936.3 2257.31  4942.5 2251.47  4947.8 2252.04  4954.4 2248.58
  4983.8 2245.31  4990.9 2244.01  4991.4 2243.51  4996.5 2244.01  5018.3 2247.84
  5038.0 2248.70  5046.6 2252.06  5081.8 2253.98  5252.8 2256.04  5387.1 2265.24
  5401.5 2264.05  5407.9 2265.39  5415.9 2263.58  5422.3 2266.03  5430.2 2262.94
  5458.9 2269.41  5494.2 2271.65  5522.9 2277.59  5529.4 2276.57  5540.7 2278.08
#Mann=6,-1,0
  4505.4   0.035       0  4618.3    0.07       0  4780.2   0.035       0
  4983.8    0.07       0  4990.9    0.07       0  4996.5    0.07       0
Bank Sta=4990.9,4996.5
Exp/Cntr=0.3,0.1

Type RM Length L Ch R = 1,12870,450,450,450
BEGIN DESCRIPTION:
UCFB HW Trib 16 27.0
END DESCRIPTION:
XS GIS Cut Line= 3
      1291171.30      6941528.58      1291755.00      6941188.00
      1291980.00      6940963.00
#Sta/Elev= 30
  4323.7 2269.52  4430.6 2266.20  4515.4 2261.98  4530.2 2261.65  4590.6 2259.22
  4649.3 2255.42  4713.8 2255.77  4729.5 2254.57  4751.0 2254.76  4756.8 2255.74
  4768.9 2254.03  4815.5 2252.03  4837.4 2252.15  4869.8 2250.03  4883.7 2249.33
  4889.9 2248.08  4895.7 2249.04  4911.4 2245.92  4964.4 2244.07  4976.3 2241.06
  4985.9 2240.92  4993.8 2237.89  4994.3 2237.39  4999.5 2237.89  5027.8 2239.42
  5056.1 2248.47  5070.2 2255.36  5155.1 2261.82  5211.6 2267.74  5317.7 2273.22
#Mann=8,-1,0
  4323.7   0.035       0  4430.6    0.07       0  4515.4   0.035       0
  4530.2    0.07       0  4768.9   0.035       0  4869.8    0.07       0
  4993.8    0.07       0  4999.5    0.07       0
Bank Sta=4993.8,4999.5
Exp/Cntr=0.3,0.1

Type RM Length L Ch R = 1,12420,465,465,465
BEGIN DESCRIPTION:
UCFB HW Trib 16 26.0
END DESCRIPTION:
XS GIS Cut Line= 3
      1291685.66      6941869.26      1292005.00      6941538.00
      1292343.17      6941053.34
#Sta/Elev= 30
  4540.1 2263.03  4596.5 2261.11  4604.7 2260.42  4745.6 2257.86  4774.0 2257.25
  4887.6 2251.81  4922.4 2248.60  4950.7 2241.72  4964.8 2239.75  4986.2 2238.50
  4996.8 2236.35  5003.3 2236.35  5010.9 2232.85  5011.3 2232.35  5016.6 2232.85
  5047.2 2236.00  5058.2 2239.16  5064.3 2239.89  5073.1 2244.81  5079.2 2243.99
  5085.6 2245.92  5094.0 2246.34  5207.5 2249.56  5293.8 2253.95  5344.4 2252.86
  5374.0 2253.87  5409.8 2253.83  5415.9 2255.64  5466.5 2256.58  5591.2 2262.92
#Mann=8,-1,0
  4540.1   0.035       0  4596.5    0.07       0  4604.7   0.035       0
  4745.6    0.07       0  4887.6   0.035       0  5010.9   0.035       0
  5016.6   0.035       0  5047.2    0.07       0
Bank Sta=5010.9,5016.6
Exp/Cntr=0.3,0.1

Type RM Length L Ch R = 1,11955,481,481,481
BEGIN DESCRIPTION:
UCFB HW Trib 16 25.0
END DESCRIPTION:
XS GIS Cut Line= 3
      1292308.48      6942047.22      1292405.00      6941738.00
      1292566.73      6941074.97
#Sta/Elev= 30
  4676.4 2264.55  4707.0 2259.54  4744.1 2257.02  4784.3 2255.83  4843.2 2252.30
  4864.1 2249.11  4881.4 2251.00  4886.6 2253.94  4906.0 2252.25  4927.0 2248.90
  4958.4 2236.11  4978.8 2233.70  4989.9 2226.80  4994.8 2226.71  4995.3 2226.21
  5000.6 2226.71  5031.2 2228.22  5060.3 2234.37  5072.4 2240.20  5165.0 2246.68
  5185.3 2247.71  5257.7 2245.42  5268.0 2240.48  5273.9 2245.57  5288.5 2245.90
  5309.1 2242.88  5315.5 2245.39  5340.0 2247.94  5445.7 2251.75  5682.8 2266.96
#Mann=5,-1,0
  4676.4    0.07       0  4744.1   0.035       0  4784.3    0.07       0
  4994.8    0.07       0  5000.6    0.07       0
Bank Sta=4994.8,5000.6
Exp/Cntr=0.3,0.1

Type RM Length L Ch R = 1,11474,469,469,469
BEGIN DESCRIPTION:
UCFB HW Trib 16 24.0
END DESCRIPTION:
XS GIS Cut Line= 3
      1292709.96      6942236.02      1292855.00      6941838.00
      1292996.41      6941407.03
#Sta/Elev= 30
  4580.3 2249.88  4612.5 2248.02  4684.6 2246.68  4810.6 2242.09  4815.9 2240.92
  4846.4 2239.82  4854.9 2238.41  4877.0 2238.23  4927.5 2235.52  4950.7 2231.75
  4972.0 2224.32  4998.3 2220.62  4998.8 2220.12  5004.2 2220.62  5051.7 2228.75
  5056.9 2227.08  5083.5 2233.50  5130.2 2239.48  5147.1 2244.15  5210.8 2246.22
  5256.5 2249.40  5288.1 2253.16  5369.9 2256.79  5401.7 2260.02  5407.0 2263.24
  5414.4 2265.29  5433.5 2266.64  5438.8 2269.27  5454.4 2263.86  5457.5 2263.86
#Mann=3,-1,0
  4580.3    0.07       0  4998.3    0.07       0  5004.2    0.07       0
Bank Sta=4998.3,5004.2
Exp/Cntr=0.3,0.1

Type RM Length L Ch R = 1,11005,452,452,452
BEGIN DESCRIPTION:
UCFB HW Trib 16 23.0
END DESCRIPTION:
XS GIS Cut Line= 5
      1292728.36      6942340.11      1293141.38      6942229.52
      1293205.00      6942138.00      1293250.75      6942069.80
      1293236.17      6941553.66
#Sta/Elev= 30
  4461.0 2250.11  4600.9 2242.28  4680.9 2239.33  4841.1 2236.05  4942.0 2235.75
  4963.5 2232.36  4971.7 2227.71  4977.8 2217.94  4989.6 2215.48  4990.1 2214.98
  4995.6 2215.48  5028.5 2218.52  5043.5 2221.47  5082.2 2225.48  5094.0 2225.73
  5103.9 2227.18  5108.9 2226.31  5134.0 2230.25  5154.0 2230.40  5174.0 2233.48
  5244.0 2238.57  5264.0 2237.95  5344.1 2239.72  5364.1 2241.26  5374.1 2240.79
  5404.1 2243.20  5424.1 2243.21  5554.1 2249.42  5574.2 2252.23  5598.5 2253.39
#Mann=3,-1,0
  4461.0    0.07       0  4989.6    0.07       0  4995.6    0.07       0
Bank Sta=4989.6,4995.6
Exp/Cntr=0.3,0.1

Type RM Length L Ch R = 1,10553,416,416,416
BEGIN DESCRIPTION:
UCFB HW Trib 16 22.0
END DESCRIPTION:
XS GIS Cut Line= 3
      1293448.05      6942434.74      1293605.00      6942288.00
      1293913.25      6941907.82
#Sta/Elev= 30
  4784.7 2230.29  4801.5 2230.13  4808.3 2230.78  4815.6 2230.07  4822.5 2231.02
  4829.8 2229.92  4872.3 2229.25  4935.8 2225.01  4964.1 2221.55  4978.3 2217.89
  4985.6 2213.57  4993.1 2211.28  4993.6 2210.78  4998.7 2210.78  4999.2 2211.28
  5013.2 2212.85  5027.6 2216.11  5041.9 2221.19  5063.9 2226.30  5070.7 2226.75
  5077.1 2226.21  5120.3 2228.05  5134.6 2230.14  5184.2 2232.99  5205.5 2234.85
  5269.9 2235.83  5283.3 2235.51  5312.1 2237.03  5347.3 2236.63  5489.0 2239.42
#Mann=3,-1,0
  4784.7    0.07       0  4993.1    0.07       0  4999.2    0.07       0
Bank Sta=4993.1,4999.2
Exp/Cntr=0.3,0.1

Type RM Length L Ch R = 1,10137,435,435,435
BEGIN DESCRIPTION:
UCFB HW Trib 16 21.0
END DESCRIPTION:
XS GIS Cut Line= 3
      1293113.74      6942592.71      1293605.00      6942638.00
      1293981.80      6942644.76
#Sta/Elev= 30
  4501.7 2233.68  4663.6 2230.31  4703.8 2232.09  4733.9 2230.21  4764.1 2230.32
  4794.2 2228.94  4854.4 2228.14  4884.6 2226.05  4904.7 2225.89  4914.7 2226.50
  4934.8 2223.87  4945.2 2220.11  4954.9 2220.06  4964.9 2217.81  4975.0 2214.52
  4992.5 2210.53  4997.5 2210.53  5012.0 2207.03  5012.5 2206.53  5017.6 2206.53
  5018.1 2207.03  5025.0 2209.51  5045.0 2212.81  5085.1 2217.80  5095.1 2222.26
  5105.1 2224.45  5145.1 2229.49  5195.1 2231.27  5255.1 2231.34  5371.9 2229.19
#Mann=3,-1,0
  4501.7    0.07       0  5012.0    0.07       0  5018.1    0.07       0
Bank Sta=5012,5018.1
Exp/Cntr=0.3,0.1

Type RM Length L Ch R = 1,9702,446,446,446
BEGIN DESCRIPTION:
UCFB HW Trib 16 20.0
END DESCRIPTION:
XS GIS Cut Line= 3
      1293230.01      6943113.00      1293605.00      6943038.00
      1293920.50      6942798.87
#Sta/Elev= 30
  4617.9 2230.02  4653.6 2228.76  4663.8 2229.42  4684.2 2227.81  4765.8 2225.52
  4776.0 2226.50  4816.7 2225.70  4891.3 2225.80  4918.7 2225.37  4939.1 2220.67
  4949.3 2211.78  4959.5 2204.80  5004.5 2203.59  5005.0 2203.09  5010.6 2203.59
  5022.1 2206.42  5028.4 2205.94  5057.5 2213.17  5078.3 2216.58  5086.6 2215.93
  5092.9 2216.77  5100.7 2216.26  5107.4 2217.44  5157.4 2219.45  5163.6 2220.39
  5201.0 2221.31  5222.4 2223.90  5263.8 2225.31  5321.7 2225.73  5396.2 2227.54
#Mann=5,-1,0
  4617.9    0.07       0  4891.3    0.16       0  5004.5    0.07       0
  5010.6    0.16       0  5222.4    0.07       0
Bank Sta=5004.5,5010.6
Exp/Cntr=0.3,0.1

Type RM Length L Ch R = 1,9256,246,246,246
BEGIN DESCRIPTION:
UCFB HW Trib 16 19.0
END DESCRIPTION:
XS GIS Cut Line= 3
      1293930.01      6943412.96      1293955.00      6943288.00
      1293979.09      6943058.90
#Sta/Elev= 30
  4872.9 2217.39  4898.4 2215.57  4908.6 2214.38  4918.8 2211.41  4929.0 2206.00
  4939.1 2204.33  4959.5 2197.20  4969.7 2196.82  4990.1 2196.95  4994.7 2196.67
  4995.2 2196.17  5000.4 2196.17  5000.9 2196.67  5051.9 2196.96  5060.7 2198.09
  5070.7 2198.97  5080.8 2201.63  5090.8 2203.42  5100.9 2203.89  5110.9 2205.23
  5139.9 2212.93  5144.9 2212.72  5151.2 2214.85  5161.2 2216.25  5171.3 2216.52
  5181.3 2216.19  5191.4 2219.15  5201.4 2220.01  5211.5 2220.11  5230.7 2220.92
#Mann=3,-1,0
  4872.9    0.07       0  4994.7    0.07       0  5000.9    0.07       0
Bank Sta=4994.7,5000.9
Exp/Cntr=0.3,0.1

Type RM Length L Ch R = 1,9010,206,206,206
BEGIN DESCRIPTION:
UCFB HW Trib 16 18.5
END DESCRIPTION:
XS GIS Cut Line= 2
      1294030.03      6943512.97      1294324.48      6943240.17
#Sta/Elev= 30
  4823.1 2217.43  4879.8 2215.93  4908.1 2212.55  4914.9 2209.92  4922.3 2205.27
  4929.1 2193.15  4947.5 2192.31  4948.0 2191.81  4953.8 2192.31  4971.6 2202.18
  4979.0 2202.22  4985.8 2198.46  4993.1 2200.91  5000.0 2197.23  5007.1 2200.39
  5014.1 2201.66  5028.3 2200.23  5035.1 2201.22  5042.5 2197.54  5049.3 2200.63
  5070.8 2199.78  5077.6 2203.05  5091.8 2206.72  5099.2 2207.57  5106.0 2209.93
  5113.3 2209.66  5120.2 2212.67  5155.9 2214.45  5162.7 2215.94  5224.5 2221.09
#Mann=3,-1,0
  4823.1    0.07       0  4947.5    0.07       0  4953.8    0.07       0
Bank Sta=4947.5,4953.8
Exp/Cntr=0.3,0.1

Type RM Length L Ch R = 1,8804,453,453,453
BEGIN DESCRIPTION:
UCFB HW Trib 16 18.0
END DESCRIPTION:
XS GIS Cut Line= 3
      1294180.01      6943612.99      1294305.00      6943538.00
      1294447.89      6943426.66
#Sta/Elev= 30
  4854.5 2214.85  4870.0 2214.97  4907.0 2211.47  4928.3 2205.87  4934.2 2205.67
  4941.9 2202.50  4949.7 2198.29  4955.6 2196.03  4965.3 2193.71  4976.9 2189.01
  4986.7 2187.31  5018.8 2186.85  5019.3 2186.35  5024.6 2186.35  5025.1 2186.85
  5028.3 2189.00  5036.4 2190.06  5042.8 2194.25  5050.9 2194.60  5057.3 2197.03
  5071.7 2199.02  5086.2 2199.24  5092.5 2201.03  5107.0 2203.73  5121.5 2207.98
  5127.8 2208.77  5136.0 2211.99  5142.3 2211.92  5156.8 2214.67  5181.4 2214.15
#Mann=3,-1,0
  4854.5    0.07       0  5018.8    0.07       0  5025.1    0.07       0
Bank Sta=5018.8,5025.1
Exp/Cntr=0.3,0.1

Type RM Length L Ch R = 1,8351,466,466,466
BEGIN DESCRIPTION:
UCFB HW Trib 16 17.0
END DESCRIPTION:
XS GIS Cut Line= 3
      1294585.12      6944267.20      1294705.00      6943688.00
      1294751.79      6943147.40
#Sta/Elev= 30
  4408.5 2222.55  4583.5 2215.70  4628.6 2212.51  4723.9 2209.39  4774.1 2205.04
  4836.6 2202.13  4857.0 2199.38  4879.6 2198.50  4897.9 2193.05  4908.1 2192.02
  4924.7 2187.53  4929.8 2188.65  4959.1 2184.04  4989.8 2183.71  5005.7 2182.18
  5006.2 2181.68  5014.4 2182.18  5030.1 2186.69  5040.1 2191.63  5056.6 2196.23
  5061.6 2195.80  5100.4 2202.35  5140.5 2206.75  5169.8 2207.72  5180.7 2205.17
  5190.7 2205.37  5210.8 2207.93  5250.9 2210.31  5361.3 2213.59  5542.6 2221.07
#Mann=3,-1,0
  4408.5    0.07       0  5005.7    0.07       0  5014.4    0.07       0
Bank Sta=5005.7,5014.4
Exp/Cntr=0.3,0.1

Type RM Length L Ch R = 1,7885,466,466,466
BEGIN DESCRIPTION:
UCFB HW Trib 16 16.0
END DESCRIPTION:
XS GIS Cut Line= 3
      1295132.00      6944374.01      1295155.00      6943738.00
      1295168.46      6943264.61
#Sta/Elev= 30
  4363.6 2212.16  4479.7 2203.15  4539.7 2200.44  4584.9 2195.30  4619.8 2194.49
  4639.8 2190.11  4649.8 2194.50  4693.3 2196.95  4732.5 2200.42  4769.9 2203.06
  4879.9 2204.88  4920.0 2199.99  4940.0 2184.29  4950.0 2181.23  4985.1 2178.63
  4985.6 2178.13  4994.9 2178.63  5010.0 2179.37  5020.0 2182.99  5030.0 2184.07
  5060.0 2180.75  5090.1 2180.58  5110.1 2189.54  5120.1 2192.35  5160.1 2196.11
  5180.5 2201.02  5210.1 2201.45  5290.1 2206.72  5430.2 2220.32  5473.6 2221.40
#Mann=5,-1,0
  4363.6    0.07       0  4693.3    0.16       0  4732.5    0.07       0
  4985.1    0.07       0  4994.9    0.07       0
Bank Sta=4985.1,4994.9
Exp/Cntr=0.3,0.1

Type RM Length L Ch R = 1,7419,445,445,445
BEGIN DESCRIPTION:
UCFB HW Trib 16 15.0
END DESCRIPTION:
XS GIS Cut Line= 3
      1295379.40      6944386.97      1295605.00      6943788.00
      1295725.18      6943461.46
#Sta/Elev= 30
  4359.9 2208.96  4478.4 2200.83  4487.0 2199.04  4583.2 2190.47  4588.5 2188.47
  4604.6 2187.04  4618.8 2182.69  4625.9 2186.43  4668.5 2190.10  4673.8 2189.43
  4679.4 2190.74  4759.1 2190.00  4814.2 2191.36  4893.1 2191.33  4935.8 2180.27
  4960.0 2178.01  4978.6 2178.35  5004.9 2175.50  5005.4 2175.00  5014.7 2175.50
  5031.9 2177.85  5045.6 2191.49  5070.8 2197.36  5076.1 2200.05  5085.2 2200.11
  5095.8 2202.05  5101.2 2204.47  5126.4 2206.50  5131.7 2205.15  5347.9 2215.22
#Mann=3,-1,0
  4359.9    0.07       0  5004.9    0.07       0  5014.7    0.07       0
Bank Sta=5004.9,5014.7
Exp/Cntr=0.3,0.1

Type RM Length L Ch R = 1,6974,481,481,481
BEGIN DESCRIPTION:
UCFB HW Trib 16 14.0
END DESCRIPTION:
XS GIS Cut Line= 3
      1295486.18      6944457.28      1295805.00      6944138.00
      1296207.54      6943728.11
#Sta/Elev= 30
  4544.0 2212.41  4556.8 2210.05  4613.4 2205.97  4634.6 2205.87  4684.1 2201.49
  4719.4 2200.12  4726.5 2198.09  4733.6 2198.17  4783.1 2192.52  4867.9 2188.12
  4889.1 2185.41  4931.6 2182.46  4945.7 2180.69  4959.9 2177.47  4981.1 2175.09
  4986.5 2173.07  4987.0 2172.57  4996.8 2173.07  5016.4 2173.39  5023.4 2175.38
  5037.6 2177.41  5065.9 2179.02  5115.4 2190.91  5136.6 2191.45  5157.9 2193.93
  5200.3 2194.96  5235.6 2194.20  5256.9 2195.62  5362.9 2197.42  5569.7 2207.85
#Mann=3,-1,0
  4544.0    0.07       0  4986.5    0.07       0  4996.8    0.07       0
Bank Sta=4986.5,4996.8
Exp/Cntr=0.3,0.1

Type RM Length L Ch R = 1,6493,485,485,485
BEGIN DESCRIPTION:
UCFB HW Trib 16 13.0
END DESCRIPTION:
XS GIS Cut Line= 3
      1296124.19      6944853.11      1296205.00      6944338.00
      1296236.06      6943821.14
#Sta/Elev= 30
  4478.6 2204.45  4666.0 2197.15  4696.3 2195.35  4736.8 2194.88  4787.4 2192.29
  4835.8 2191.26  4848.2 2188.60  4858.3 2184.23  4888.7 2184.94  4898.5 2183.80
  4903.5 2184.86  4908.9 2182.70  4929.2 2179.34  4979.8 2175.89  4989.9 2172.74
  4992.3 2169.38  4992.8 2168.88  5002.7 2169.38  5010.0 2170.69  5070.1 2174.82
  5079.3 2176.09  5084.3 2175.30  5090.2 2177.27  5110.2 2176.65  5150.3 2177.48
  5180.3 2179.24  5260.5 2190.32  5290.5 2192.53  5470.9 2200.92  5517.8 2203.95
#Mann=3,-1,0
  4478.6    0.07       0  4992.3    0.07       0  5002.7    0.07       0
Bank Sta=4992.3,5002.7
Exp/Cntr=0.3,0.1

Type RM Length L Ch R = 1,6008,472,472,472
BEGIN DESCRIPTION:
UCFB HW Trib 16 12.0
END DESCRIPTION:
XS GIS Cut Line= 3
      1296478.35      6944907.83      1296655.00      6944338.00
      1296710.06      6943994.16
#Sta/Elev= 30
  4402.8 2200.70  4511.1 2194.68  4664.4 2188.83  4842.3 2186.53  4852.8 2183.11
  4885.3 2176.05  4917.9 2175.09  4926.1 2173.57  4945.3 2172.52  4957.5 2170.36
  4977.8 2171.12  4996.8 2167.72  5027.8 2167.47  5034.7 2166.13  5035.2 2165.63
  5045.1 2166.13  5050.0 2166.17  5060.1 2172.86  5070.3 2175.65  5120.9 2182.63
  5131.0 2182.45  5141.2 2186.37  5156.9 2190.00  5181.7 2192.04  5224.0 2193.44
  5272.8 2196.28  5280.9 2197.61  5303.2 2198.22  5342.9 2202.12  5347.6 2201.39
#Mann=3,-1,0
  4402.8    0.07       0  5034.7    0.07       0  5045.1    0.07       0
Bank Sta=5034.7,5045.1
Exp/Cntr=0.3,0.1

Type RM Length L Ch R = 1,5536,435,435,435
BEGIN DESCRIPTION:
UCFB HW Trib 16 11.0
END DESCRIPTION:
XS GIS Cut Line= 3
      1296863.77      6945053.67      1296955.00      6944638.00
      1297048.67      6944163.01
#Sta/Elev= 30
  4574.6 2214.37  4599.7 2212.90  4621.4 2207.66  4653.7 2204.12  4682.8 2203.61
  4713.5 2200.85  4723.7 2201.39  4741.3 2199.30  4790.3 2196.02  4795.4 2194.94
  4856.8 2190.73  4883.0 2187.72  4888.1 2188.75  4897.8 2188.04  4918.3 2183.48
  4926.8 2178.09  4931.9 2177.51  4938.7 2172.13  4959.2 2166.99  4970.5 2162.08
  4971.0 2161.58  4981.0 2162.08  5002.7 2164.01  5020.5 2167.11  5025.8 2169.02
  5051.1 2172.83  5071.5 2174.47  5142.9 2183.57  5163.2 2184.81  5484.3 2185.58
#Mann=3,-1,0
  4574.6    0.07       0  4970.5    0.07       0  4981.0    0.07       0
Bank Sta=4970.5,4981
Exp/Cntr=0.3,0.1

Type RM Length L Ch R = 1,5101,460,460,460
BEGIN DESCRIPTION:
UCFB HW Trib 16 10.0
END DESCRIPTION:
XS GIS Cut Line= 3
      1297197.10      6945048.47      1297305.00      6944738.00
      1297415.85      6944347.93
#Sta/Elev= 30
  4663.3 2203.72  4666.2 2203.72  4675.9 2200.36  4695.6 2198.54  4716.7 2194.09
  4748.5 2190.37  4852.0 2184.71  4896.7 2183.78  4928.5 2181.86  4939.1 2180.20
  4950.6 2175.88  4960.2 2173.70  4970.8 2170.01  4976.4 2164.87  4981.7 2164.91
  4989.3 2158.90  4997.1 2158.18  4997.6 2157.68  5007.7 2158.18  5014.1 2158.34
  5023.2 2161.42  5033.6 2168.23  5042.8 2170.26  5081.9 2173.75  5087.1 2173.40
  5115.8 2176.57  5127.1 2179.37  5147.9 2182.35  5379.0 2181.20  5397.5 2181.74
#Mann=3,-1,0
  4663.3    0.07       0  4997.1    0.07       0  5007.7    0.07       0
Bank Sta=4997.1,5007.7
Exp/Cntr=0.3,0.1

Type RM Length L Ch R = 1,4641,479,479,479
BEGIN DESCRIPTION:
UCFB HW Trib 16 9.0
END DESCRIPTION:
XS GIS Cut Line= 3
      1297353.38      6945176.02      1297755.00      6944688.00
      1297930.01      6944562.99
#Sta/Elev= 30
  4371.9 2194.05  4541.9 2184.15  4628.0 2181.20  4712.7 2180.49  4770.0 2177.62
  4840.4 2172.37  4869.1 2172.42  4889.9 2171.39  4932.9 2167.85  4953.7 2164.58
  4961.6 2161.02  4968.1 2161.70  4975.9 2157.34  4991.4 2155.38  4991.9 2154.88
  5002.1 2155.38  5003.9 2156.94  5011.3 2158.39  5017.4 2158.12  5026.0 2165.85
  5032.2 2159.35  5040.8 2163.42  5067.8 2169.46  5076.4 2170.12  5089.9 2172.71
  5097.3 2175.10  5103.5 2174.94  5112.1 2176.93  5176.0 2178.67  5219.0 2178.24
#Mann=3,-1,0
  4371.9    0.07       0  4991.4    0.07       0  5002.1    0.07       0
Bank Sta=4991.4,5002.1
Exp/Cntr=0.3,0.1

Type RM Length L Ch R = 1,4162,472,472,472
BEGIN DESCRIPTION:
UCFB HW Trib 16 8.0
END DESCRIPTION:
XS GIS Cut Line= 3
      1297530.02      6945312.98      1297755.00      6945138.00
      1297930.02      6945012.99
#Sta/Elev= 30
  4711.0 2188.04  4781.6 2183.57  4796.0 2183.53  4804.2 2182.84  4810.5 2183.22
  4839.5 2181.46  4874.8 2180.73  4882.0 2179.95  4953.5 2179.08  4959.8 2176.15
  4968.0 2170.98  4982.4 2157.86  4988.8 2155.97  4992.9 2153.74  4998.0 2153.41
  4998.5 2152.91  5008.2 2152.91  5008.7 2153.41  5032.9 2157.90  5045.2 2162.52
  5053.8 2164.29  5068.5 2164.40  5095.6 2167.42  5104.2 2170.78  5110.3 2170.22
  5118.9 2172.20  5145.9 2176.90  5168.1 2178.27  5196.3 2178.54  5211.1 2177.82
#Mann=3,-1,0
  4711.0    0.07       0  4998.0    0.07       0  5008.7    0.07       0
Bank Sta=4998,5008.7
Exp/Cntr=0.3,0.1

Type RM Length L Ch R = 1,3690,465,465,465
BEGIN DESCRIPTION:
UCFB HW Trib 16 7.0
END DESCRIPTION:
XS GIS Cut Line= 3
      1297980.03      6945512.97      1298155.00      6945338.00
      1298130.00      6945263.01
#Sta/Elev= 29
  4760.5 2175.15  4781.7 2175.69  4795.8 2175.87  4810.0 2175.64  4824.1 2175.22
  4838.2 2174.69  4852.4 2173.93  4880.7 2173.05  4894.8 2172.88  4909.0 2172.93
  4923.1 2172.09  4937.2 2169.78  4951.4 2166.35  4965.5 2162.78  4979.7 2150.95
  4988.5 2150.02  4989.0 2149.52  4998.7 2149.52  4999.2 2150.02  5004.4 2154.25
  5010.6 2154.25  5018.5 2161.62  5029.0 2162.81  5039.6 2163.20  5050.1 2163.77
  5060.7 2163.90  5071.2 2165.13  5081.7 2164.50  5087.0 2164.50
#Mann=3,-1,0
  4760.5    0.07       0  4988.5    0.07       0  4999.2    0.07       0
Bank Sta=4988.5,4999.2
Exp/Cntr=0.3,0.1

Type RM Length L Ch R = 1,3225,479,479,479
BEGIN DESCRIPTION:
UCFB HW Trib 16 6.0
END DESCRIPTION:
XS GIS Cut Line= 3
      1298255.00      6945788.00      1298505.00      6945588.00
      1298596.96      6945506.26
#Sta/Elev= 30
  4683.9 2172.65  4705.5 2171.72  4726.3 2165.95  4755.1 2162.18  4761.5 2159.05
  4769.5 2159.07  4775.9 2155.63  4784.0 2155.66  4790.4 2153.02  4833.6 2153.03
  4848.0 2154.14  4854.4 2156.72  4862.4 2154.52  4876.0 2153.54  4932.8 2154.64
  4982.4 2149.43  4983.2 2148.28  4983.7 2147.78  4997.7 2148.28  5000.9 2152.12
  5007.4 2152.12  5011.2 2159.18  5017.9 2164.05  5025.4 2171.73  5053.8 2171.11
  5060.5 2169.70  5068.0 2171.07  5074.7 2169.00  5096.5 2170.70  5127.1 2169.33
#Mann=3,-1,0
  4683.9    0.07       0  4983.2    0.07       0  4997.7    0.07       0
Bank Sta=4983.2,4997.7
Exp/Cntr=0.3,0.1

Type RM Length L Ch R = 1,2746,455,455,455
BEGIN DESCRIPTION:
UCFB HW Trib 16 5.0
END DESCRIPTION:
XS GIS Cut Line= 3
      1298428.99      6946039.15      1298605.00      6946038.00
      1298804.99      6946038.00
#Sta/Elev= 30
  4824.0 2171.08  4840.0 2171.17  4860.0 2170.93  4870.0 2169.88  4890.0 2164.86
  4900.0 2163.93  4910.0 2162.40  4920.0 2158.20  4930.0 2155.15  4940.0 2152.55
  4950.0 2152.85  4960.0 2152.33  4970.0 2150.72  4980.0 2148.57  4990.0 2147.28
  4990.3 2146.38  4990.8 2145.88  5004.3 2145.88  5004.8 2146.38  5010.0 2149.32
  5020.0 2157.53  5030.0 2167.42  5040.0 2169.51  5050.0 2169.58  5070.0 2170.23
  5100.0 2170.46  5120.0 2170.10  5140.0 2169.34  5180.0 2168.96  5200.0 2169.13
#Mann=3,-1,0
  4824.0    0.07       0  4990.3    0.07       0  5004.8    0.07       0
Bank Sta=4990.3,5004.8
Exp/Cntr=0.3,0.1

Type RM Length L Ch R = 1,2291,220,220,220
BEGIN DESCRIPTION:
UCFB HW Trib 16 4.0
END DESCRIPTION:
XS GIS Cut Line= 2
      1298734.56      6946369.00      1298975.84      6946296.96
#Sta/Elev= 30
  4838.2 2168.71  4841.0 2168.71  4849.1 2168.22  4862.0 2167.94  4870.0 2167.58
  4880.4 2166.97  4889.9 2166.09  4895.1 2162.25  4901.3 2159.63  4911.7 2155.01
  4922.1 2152.59  4933.4 2150.23  4943.0 2149.00  4961.4 2147.19  4966.6 2147.71
  4974.3 2146.83  4984.8 2143.75  4987.2 2143.31  4987.7 2142.81  5001.3 2142.81
  5001.8 2143.31  5005.6 2150.38  5016.1 2159.88  5026.5 2168.71  5032.8 2168.38
  5057.8 2168.42  5066.0 2168.24  5071.2 2168.35  5078.7 2168.37  5090.0 2168.20
#Mann=3,-1,0
  4838.2    0.07       0  4987.2    0.07       0  5001.8    0.07       0
Bank Sta=4987.2,5001.8
Exp/Cntr=0.3,0.1

Type RM Length L Ch R = 1,2071,180,180,180
BEGIN DESCRIPTION:
UCFB HW Trib 16 3.3
END DESCRIPTION:
XS GIS Cut Line= 2
      1298895.10      6946604.26      1299094.76      6946416.76
#Sta/Elev= 30
  4850.7 2167.61  4855.0 2167.99  4862.3 2167.87  4869.1 2167.27  4876.4 2167.07
  4890.6 2164.87  4897.5 2162.97  4904.8 2161.50  4918.9 2159.34  4932.9 2158.33
  4940.0 2158.52  4946.8 2157.70  4954.1 2157.63  4961.0 2152.96  4968.3 2150.20
  4975.1 2142.81  4975.6 2142.31  4989.2 2142.31  4989.7 2142.81  5003.5 2153.72
  5010.8 2158.85  5017.6 2162.72  5024.9 2165.16  5031.8 2164.69  5039.1 2165.68
  5046.0 2165.20  5053.3 2165.71  5074.3 2165.31  5095.8 2164.36  5124.6 2163.70
#Mann=3,-1,0
  4850.7    0.07       0  4975.1    0.07       0  4989.7    0.07       0
Bank Sta=4975.1,4989.7
Exp/Cntr=0.3,0.1

Type RM Length L Ch R = 1,1891,166,166,166
BEGIN DESCRIPTION:
UCFB HW Trib 16 3.15
END DESCRIPTION:
XS GIS Cut Line= 2
      1299022.70      6946739.69      1299168.56      6946572.99
#Sta/Elev= 30
  4869.6 2167.19  4874.1 2167.19  4879.6 2167.55  4886.2 2165.92  4893.8 2164.87
  4900.5 2161.15  4908.1 2159.86  4914.7 2158.04  4928.9 2156.17  4943.2 2155.24
  4950.8 2154.95  4957.4 2151.94  4964.9 2152.62  4978.3 2144.75  4978.6 2142.51
  4979.1 2142.01  4992.7 2142.01  4993.2 2142.51  5000.1 2144.90  5006.8 2148.58
  5014.4 2152.53  5021.0 2160.41  5028.6 2162.24  5035.2 2162.52  5042.8 2163.10
  5049.5 2162.85  5057.1 2163.78  5063.7 2163.68  5071.2 2163.96  5091.1 2164.05
#Mann=3,-1,0
  4869.6    0.07       0  4978.6    0.07       0  4993.2    0.07       0
Bank Sta=4978.6,4993.2
Exp/Cntr=0.3,0.1

Type RM Length L Ch R = 1,1725,91,91,91
BEGIN DESCRIPTION:
UCFB HW Trib 16 3.2
END DESCRIPTION:
XS GIS Cut Line= 4
      1299130.01      6946862.99      1299174.77      6946780.38
      1299239.87      6946759.77      1299227.95      6946688.20
#Sta/Elev= 30
  4873.7 2165.83  4879.4 2165.68  4889.9 2166.31  4895.6 2166.12  4902.1 2165.11
  4911.7 2161.91  4917.4 2160.59  4924.9 2157.57  4933.6 2156.69  4939.3 2154.42
  4947.6 2152.49  4955.5 2151.12  4961.2 2148.34  4966.2 2147.10  4970.4 2147.10
  4978.4 2145.12  4985.8 2143.53  4986.3 2143.03  4999.9 2143.03  5000.4 2143.53
  5009.9 2145.70  5020.2 2147.80  5025.4 2150.71  5030.8 2154.11  5039.4 2154.11
  5047.9 2157.39  5058.0 2157.92  5068.2 2158.21  5088.4 2159.85  5108.5 2160.34
#Mann=3,-1,0
  4873.7    0.07       0  4985.8    0.07       0  5000.4    0.07       0
Bank Sta=4985.8,5000.4
Exp/Cntr=0.3,0.1

Type RM Length L Ch R = 1,1634,156,156,156
BEGIN DESCRIPTION:
UCFB HW Trib 16 3.1
END DESCRIPTION:
XS GIS Cut Line= 3
      1299262.76      6946947.75      1299260.03      6946742.82
      1299229.14      6946688.31
#Sta/Elev= 30
  4888.5 2164.54  4890.9 2164.54  4898.3 2164.25  4908.3 2164.35  4918.3 2164.79
  4928.3 2157.34  4938.3 2151.10  4948.3 2149.22  4958.3 2146.86  4968.3 2143.30
  4971.0 2143.11  4971.5 2142.61  4985.1 2142.61  4985.6 2143.11  4988.3 2144.05
  5008.3 2145.31  5018.3 2146.47  5028.3 2148.16  5048.3 2152.78  5058.3 2156.52
  5078.3 2157.01  5088.3 2157.35  5099.1 2157.94  5109.3 2157.60  5115.0 2157.97
  5122.0 2159.09  5136.6 2159.85  5145.0 2160.03  5152.5 2159.97  5156.1 2160.34
#Mann=3,-1,0
  4888.5    0.07       0  4971.0    0.07       0  4985.6    0.07       0
Bank Sta=4971,4985.6
Exp/Cntr=0.3,0.1

Type RM Length L Ch R = 1,1478,81,81,81
BEGIN DESCRIPTION:
UCFB HW Trib 16 3.05
END DESCRIPTION:
XS GIS Cut Line= 2
      1299418.36      6946808.44      1299228.88      6946685.45
#Sta/Elev= 30
  4925.1 2165.10  4935.1 2165.41  4941.1 2165.23  4956.2 2165.38  4964.9 2162.90
  4971.3 2152.20  4977.3 2151.10  4986.5 2145.26  4992.4 2144.93  5000.3 2141.60
  5000.8 2141.10  5014.4 2141.10  5014.9 2141.60  5022.7 2145.01  5028.7 2144.57
  5036.4 2146.75  5043.8 2148.42  5049.8 2149.08  5059.0 2154.22  5064.9 2154.13
  5072.2 2154.47  5080.1 2156.17  5086.0 2156.13  5095.2 2157.64  5101.2 2157.55
  5116.3 2159.11  5122.3 2159.51  5131.5 2159.74  5137.4 2159.55  5151.0 2160.34
#Mann=4,-1,0
  4925.1   0.035       0  4941.1    0.07       0  5000.3    0.07       0
  5014.9    0.07       0
Bank Sta=5000.3,5014.9
Exp/Cntr=0.3,0.1

Type RM Length L Ch R = 1,1397,180,180,180
BEGIN DESCRIPTION:
UCFB HW Trib 16 3.0
END DESCRIPTION:
XS GIS Cut Line= 3
      1299441.08      6946688.45      1299355.00      6946688.00
      1299215.04      6946679.55
#Sta/Elev= 30
  4909.2 2164.49  4915.3 2164.48  4925.3 2164.73  4935.3 2165.18  4942.1 2164.30
  4945.3 2163.89  4955.3 2161.05  4965.3 2152.96  4975.3 2146.61  4985.3 2144.23
  4992.8 2143.10  4997.8 2143.10  4998.0 2143.03  4998.5 2142.53  5012.1 2142.53
  5012.6 2143.03  5015.3 2143.89  5025.3 2145.40  5035.4 2151.12  5045.4 2153.35
  5055.4 2154.04  5065.4 2155.94  5074.3 2157.52  5079.3 2157.05  5085.4 2157.42
  5095.5 2158.41  5105.5 2159.08  5125.5 2160.11  5133.0 2160.38  5135.5 2160.38
#Mann=4,-1,0
  4909.2   0.035       0  4942.1    0.07       0  4998.0    0.07       0
  5012.6    0.07       0
Bank Sta=4998,5012.6
Exp/Cntr=0.3,0.1

Type RM Length L Ch R = 1,1217,345,345,345
BEGIN DESCRIPTION:
UCFB HW Trib 16 2.5
END DESCRIPTION:
XS GIS Cut Line= 2
      1299407.90      6946543.95      1299248.50      6946511.35
#Sta/Elev= 25
  4894.7 2160.28  4897.1 2160.28  4901.1 2160.08  4907.9 2159.05  4918.1 2156.69
  4928.3 2155.11  4938.5 2155.51  4946.5 2155.15  4951.6 2153.60  4958.9 2150.06
  4969.1 2143.64  4972.0 2141.56  4972.5 2141.06  4986.1 2141.06  4986.6 2141.56
  4989.5 2141.61  4996.9 2142.02  5002.0 2142.34  5009.9 2149.43  5020.1 2157.99
  5030.4 2163.40  5040.6 2163.59  5047.4 2163.37  5052.5 2163.91  5057.4 2163.79
#Mann=3,-1,0
  4894.7    0.07       0  4972.0    0.07       0  4986.6    0.07       0
Bank Sta=4972,4986.6
Exp/Cntr=0.3,0.1

Type RM Length L Ch R = 1,872,54,54,54
BEGIN DESCRIPTION:
UCFB HW Trib 16 2.0
END DESCRIPTION:
XS GIS Cut Line= 3
      1299505.00      6946737.97      1299525.13      6946387.45
      1299561.94      6946206.56
#Sta/Elev= 30
  4648.9 2164.46  4688.9 2164.56  4719.0 2163.55  4729.0 2162.59  4735.0 2160.69
  4740.0 2162.45  4746.5 2161.93  4759.1 2161.79  4779.1 2159.46  4869.2 2157.29
  4949.4 2156.99  4959.4 2154.09  4979.4 2145.65  5002.3 2143.86  5017.3 2141.81
  5017.8 2141.31  5031.5 2141.31  5032.0 2141.81  5040.3 2148.70  5060.7 2154.16
  5070.2 2162.48  5075.3 2160.64  5084.6 2161.82  5091.3 2162.35  5101.5 2164.50
  5111.7 2165.28  5120.7 2165.82  5125.8 2164.63  5134.4 2165.29  5184.6 2165.25
#Mann=6,-1,0
  4648.9   0.035       0  4746.5    0.07       0  5017.3    0.07       0
  5032.0    0.07       0  5084.6   0.035       0  5134.4    0.07       0
Bank Sta=5017.3,5032
Exp/Cntr=0.3,0.1

Type RM Length L Ch R = 1,818,302,302,302
BEGIN DESCRIPTION:
UCFB HW Trib 16 1.5
END DESCRIPTION:
XS GIS Cut Line= 2
      1299536.26      6946617.61      1299606.49      6946215.70
#Sta/Elev= 30
  4785.7 2162.47  4815.8 2162.93  4836.1 2162.50  4856.4 2161.05  4863.5 2159.61
  4868.6 2161.07  4876.7 2161.03  4907.1 2157.70  4947.7 2156.66  4957.9 2154.77
  4968.0 2153.37  4977.4 2149.91  4988.3 2144.81  4998.5 2142.62  5011.4 2141.45
  5011.9 2140.95  5025.6 2140.95  5026.1 2141.45  5028.9 2141.65  5032.7 2142.81
  5042.0 2145.21  5059.4 2156.52  5069.6 2159.89  5079.7 2161.23  5096.4 2161.01
  5101.5 2162.11  5143.6 2162.19  5155.9 2162.69  5161.0 2163.40  5193.7 2163.91
#Mann=5,-1,0
  4785.7    0.07       0  5011.4    0.07       0  5026.1    0.07       0
  5032.7   0.035       0  5143.6    0.07       0
Bank Sta=5011.4,5026.1
Exp/Cntr=0.3,0.1

Type RM Length L Ch R = 1,516,255,255,255
BEGIN DESCRIPTION:
UCFB HW Trib 16 1.0
END DESCRIPTION:
XS GIS Cut Line= 3
      1299712.81      6946672.54      1299805.00      6946588.00
      1299889.08      6946512.48
#Sta/Elev= 30
  4875.2 2161.69  4901.3 2161.95  4913.1 2161.53  4922.3 2160.99  4929.7 2159.00
  4936.5 2156.59  4943.9 2155.63  4950.6 2153.13  4964.8 2152.21  4972.2 2150.07
  4986.4 2147.87  4993.2 2144.67  4996.9 2141.71  5003.3 2141.71  5006.8 2140.04
  5007.3 2139.54  5021.0 2139.54  5021.5 2140.04  5021.6 2140.37  5028.3 2141.70
  5035.8 2146.50  5050.0 2153.25  5056.7 2154.70  5065.1 2154.55  5070.9 2156.09
  5078.4 2155.36  5092.6 2157.67  5099.3 2159.72  5106.8 2160.76  5113.3 2160.72
#Mann=6,-1,0
  4875.2    0.07       0  4913.1   0.035       0  5003.3    0.07       0
  5006.8   0.035       0  5021.5    0.07       0  5065.1   0.035       0
Bank Sta=5006.8,5021.5
Exp/Cntr=0.3,0.1

Type RM Length L Ch R = 1,261,0,0,0
BEGIN DESCRIPTION:
UCFB HW Trib 16 0.5
END DESCRIPTION:
XS GIS Cut Line= 3
      1300011.22      6946714.80      1300018.91      6946650.06
      1300031.83      6946523.92
#Sta/Elev= 27
  4872.5 2156.94  4879.4 2156.84  4889.4 2155.86  4899.5 2154.67  4909.6 2153.44
  4919.6 2152.74  4929.7 2152.52  4936.2 2146.25  4941.2 2146.25  4946.6 2141.08
  4951.6 2142.12  4959.9 2139.56  4962.6 2138.72  4963.1 2138.22  4976.8 2138.22
  4977.3 2138.72  4980.0 2139.07  4990.0 2141.75  5000.1 2147.67  5010.1 2149.58
  5020.2 2150.31  5030.2 2150.08  5040.3 2153.86  5045.9 2158.81  5051.0 2155.94
  5060.0 2159.25  5064.5 2159.25
#Mann=3,-1,0
  4872.5    0.07       0  4962.6    0.07       0  4977.3    0.07       0
Bank Sta=4962.6,4977.3
Exp/Cntr=0.3,0.1

Chan Stop Cuts=-1
