HEC-RAS study Bull Creek.prj: Bull Creek Base Level Engineering

--- Bull Creek.g01 (geometry) --- (continued)

Type RM Length L Ch R = 1,35000,500,500,500
BEGIN DESCRIPTION:
Bull Creek 70.0
END DESCRIPTION:
XS GIS Cut Line= 3
      1327654.99      6919038.02      1327722.00      6918921.29
      1328104.97      6918438.04
#Sta/Elev= 30
  4865.4 2161.96  4916.5 2160.81  4938.0 2158.61  4959.6 2157.93  4975.4 2151.49
  4985.5 2151.05  4986.0 2150.55  4996.9 2151.05  4997.0 2152.23  4999.0 2153.81
  5026.2 2155.68  5055.0 2156.80  5061.4 2154.40  5068.0 2156.56  5075.8 2157.54
  5082.2 2156.73  5111.1 2157.35  5119.0 2160.00  5131.9 2162.05  5139.9 2162.83
  5146.3 2161.98  5154.4 2163.84  5160.7 2163.26  5168.8 2164.58  5175.2 2164.08
  5182.8 2165.79  5361.1 2165.86  5502.0 2168.61  5559.8 2171.02  5616.6 2171.61
#Mann=3,-1,0
  4865.4   0.035       0  4985.5   0.035       0  4996.9   0.035       0
Bank Sta=4985.5,4996.9
Exp/Cntr=0.3,0.1

Type RM Length L Ch R = 1,34500,500,500,500
BEGIN DESCRIPTION:
Bull Creek 69.0
END DESCRIPTION:
XS GIS Cut Line= 3
      1326755.03      6919337.99      1327760.83      6919129.95
      1328704.95      6919188.00
#Sta/Elev= 30
  3972.9 2191.57  4198.8 2184.77  4389.5 2182.27  4439.7 2181.12  4444.8 2180.00
  4540.1 2178.84  4545.2 2177.92  4685.7 2174.80  4830.7 2166.25  4841.4 2162.77
  4851.1 2153.94  4861.3 2153.00  4875.6 2148.52  4876.1 2148.02  4887.1 2148.52
  4891.9 2150.46  4906.0 2152.10  4931.6 2153.17  4936.7 2151.59  4943.0 2154.04
  4947.9 2154.58  4986.9 2158.54  5024.2 2158.03  5074.3 2159.90  5294.7 2159.26
  5384.9 2154.15  5536.9 2158.80  5573.0 2161.12  5835.7 2172.80  5945.9 2179.95
#Mann=7,-1,0
  3972.9   0.035       0  4875.6   0.035       0  4887.1   0.035       0
  4906.0    0.07       0  4947.9   0.035       0  5536.9    0.07       0
  5573.0   0.035       0
Bank Sta=4875.6,4887.1
Exp/Cntr=0.3,0.1

Type RM Length L Ch R = 1,34000,500,500,500
BEGIN DESCRIPTION:
Bull Creek 68.0
END DESCRIPTION:
XS GIS Cut Line= 3
      1327321.12      6919523.88      1327975.63      6919358.81
      1328730.41      6919475.20
#Sta/Elev= 30
  4325.0 2200.10  4401.2 2197.68  4577.8 2186.30  4762.1 2181.57  4813.7 2175.96
  4824.2 2170.63  4876.6 2167.11  4937.1 2162.90  4942.3 2157.57  4947.8 2155.53
  4978.2 2151.67  4989.0 2148.60  4991.3 2145.94  4991.8 2145.44  5002.8 2145.94
  5026.1 2150.39  5031.1 2148.94  5070.2 2151.49  5130.9 2150.41  5162.5 2147.50
  5225.7 2150.20  5252.0 2158.00  5313.0 2172.91  5357.1 2177.87  5418.2 2190.41
  5488.5 2195.02  5614.8 2194.93  5707.6 2204.73  5738.0 2205.45  5763.7 2202.27
#Mann=6,-1,0
  4325.0   0.035       0  4876.6    0.07       0  4991.3   0.035       0
  5002.8    0.07       0  5252.0    0.07       0  5418.2   0.035       0
Bank Sta=4991.3,5002.8
Exp/Cntr=0.3,0.1

Type RM Length L Ch R = 1,33500,500,500,500
BEGIN DESCRIPTION:
Bull Creek 67.0
END DESCRIPTION:
XS GIS Cut Line= 3
      1327328.05      6919593.32      1328104.72      6919715.99
      1328779.48      6919537.76
#Sta/Elev= 30
  4213.7 2202.64  4322.0 2197.20  4524.5 2191.64  4666.2 2179.36  4853.1 2169.51
  4909.2 2162.13  4920.5 2158.30  4959.8 2151.08  4990.2 2151.18  5002.7 2148.78
  5008.6 2144.65  5013.8 2146.17  5015.1 2142.97  5015.6 2142.47  5026.9 2142.97
  5048.9 2148.96  5054.0 2148.44  5083.0 2153.46  5089.1 2156.74  5094.3 2156.76
  5124.2 2164.08  5209.9 2171.37  5285.3 2179.72  5527.8 2195.95  5556.8 2194.98
  5561.9 2196.24  5597.0 2193.99  5602.2 2195.76  5637.3 2194.35  5697.9 2196.68
#Mann=3,-1,0
  4213.7   0.035       0  5015.1   0.035       0  5026.9   0.035       0
Bank Sta=5015.1,5026.9
Exp/Cntr=0.3,0.1

Type RM Length L Ch R = 1,33000,500,500,500
BEGIN DESCRIPTION:
Bull Creek 66.0
END DESCRIPTION:
XS GIS Cut Line= 3
      1327425.26      6920329.44      1328339.67      6920088.97
      1328953.05      6919426.68
#Sta/Elev= 30
  4054.5 2191.65  4195.8 2185.44  4357.2 2183.00  4519.5 2176.25  4736.7 2163.12
  4798.7 2157.56  4825.7 2157.03  4860.8 2150.59  4891.8 2150.43  4922.8 2148.09
  4933.1 2146.73  4941.6 2142.58  4958.2 2141.56  4958.7 2141.06  4970.1 2141.56
  4981.9 2143.18  4987.1 2147.59  5004.3 2147.83  5025.8 2151.13  5032.7 2150.34
  5061.0 2152.62  5138.7 2154.19  5400.6 2168.75  5408.0 2171.43  5414.8 2175.92
  5429.0 2178.20  5436.3 2177.83  5471.5 2183.67  5782.8 2197.80  5902.7 2206.05
#Mann=3,-1,0
  4054.5   0.035       0  4958.2   0.035       0  4970.1   0.035       0
Bank Sta=4958.2,4970.1
Exp/Cntr=0.3,0.1

Type RM Length L Ch R = 1,32500,500,500,500
BEGIN DESCRIPTION:
Bull Creek 65.0
END DESCRIPTION:
XS GIS Cut Line= 3
      1327536.44      6920489.14      1328794.34      6920126.24
      1328987.78      6919405.85
#Sta/Elev= 30
  3690.8 2185.58  3970.5 2171.24  4334.6 2161.31  4361.5 2153.76  4376.2 2158.31
  4395.1 2154.38  4400.3 2158.53  4439.2 2147.93  4467.6 2155.39  4490.7 2148.64
  4506.5 2153.66  4605.2 2155.84  4796.5 2147.83  4975.1 2147.20  5008.5 2144.11
  5017.0 2139.56  5017.5 2139.06  5028.9 2139.56  5049.9 2147.62  5081.0 2151.09
  5097.7 2146.01  5137.7 2145.50  5172.5 2156.34  5177.7 2153.00  5212.5 2162.70
  5217.7 2159.58  5257.7 2159.94  5350.2 2166.28  5402.0 2184.94  5745.9 2209.23
#Mann=3,-1,0
  3690.8   0.035       0  5017.0   0.035       0  5028.9   0.035       0
Bank Sta=5017,5028.9
Exp/Cntr=0.3,0.1

Type RM Length L Ch R = 1,32000,500,500,500
BEGIN DESCRIPTION:
Bull Creek 64.0
END DESCRIPTION:
XS GIS Cut Line= 3
      1327529.47      6920489.15      1329154.85      6920410.08
      1329182.23      6919384.95
#Sta/Elev= 30
  3372.7 2185.93  3608.5 2174.25  3888.8 2164.65  4189.2 2158.29  4669.8 2154.05
  4890.0 2148.42  4950.1 2145.66  4974.2 2139.31  4974.7 2138.81  4986.1 2139.31
  4997.6 2143.59  5062.1 2145.00  5092.1 2149.32  5162.1 2151.61  5232.2 2157.49
  5292.2 2159.33  5422.2 2169.82  5472.2 2177.87  5522.3 2194.67  5552.3 2199.57
  5567.3 2205.40  5602.3 2205.72  5622.3 2208.95  5652.3 2209.89  5682.3 2207.32
  5742.3 2210.69  5783.2 2209.70  5784.7 2209.67  5952.4 2209.27  6025.5 2211.49
#Mann=5,-1,0
  3372.7   0.035       0  4974.2   0.035       0  4986.1   0.035       0
  5783.2    0.07       0  5784.7   0.035       0
Bank Sta=4974.2,4986.1
Exp/Cntr=0.3,0.1

Type RM Length L Ch R = 1,31500,500,500,500
BEGIN DESCRIPTION:
Bull Creek 63.0
END DESCRIPTION:
XS GIS Cut Line= 4
      1327564.19      6920461.38      1329339.86      6920750.15
      1329494.48      6920638.02      1329848.89      6919718.34
#Sta/Elev= 30
  3010.0 2183.54  3330.8 2170.14  3649.1 2160.19  4836.0 2149.31  4936.6 2144.06
  4942.7 2141.02  4972.1 2141.41  4986.8 2139.93  4993.0 2136.64  5002.7 2137.98
  5009.7 2136.09  5010.2 2135.59  5021.7 2136.09  5032.2 2143.99  5070.3 2146.90
  5201.9 2147.21  5248.9 2148.94  5385.8 2154.49  5433.3 2157.86  5493.2 2167.08
  5525.1 2168.10  5542.5 2170.52  5547.8 2169.44  5567.1 2172.18  5572.5 2171.42
  5691.3 2180.07  5820.8 2185.34  5850.8 2181.16  5960.6 2178.01  5985.6 2177.26
#Mann=7,-1,0
  3010.0   0.035       0  5009.7   0.035       0  5021.7   0.035       0
  5201.9    0.07       0  5248.9   0.035       0  5691.3    0.07       0
  5960.6   0.035       0
Bank Sta=5009.7,5021.7
Exp/Cntr=0.3,0.1

Type RM Length L Ch R = 1,31000,367,367,367
BEGIN DESCRIPTION:
Bull Creek 62.0
END DESCRIPTION:
XS GIS Cut Line= 4
      1327730.83      6920551.65      1329779.45      6920857.21
      1329973.35      6920605.40      1330626.69      6919794.69
#Sta/Elev= 30
  2610.9 2177.11  2928.5 2164.10  3089.9 2159.66  4162.0 2150.76  4495.7 2149.66
  4942.6 2142.33  4971.5 2141.59  4978.0 2136.59  4984.3 2138.29  4991.2 2135.76
  4991.7 2135.26  5003.4 2135.76  5035.2 2137.71  5042.0 2139.20  5048.5 2145.90
  5056.4 2143.33  5062.9 2149.06  5070.8 2146.68  5077.2 2146.74  5085.2 2147.75
  5091.6 2151.77  5099.4 2152.60  5120.4 2149.29  5163.6 2153.60  5211.5 2154.68
  5341.1 2156.91  5531.3 2164.51  5731.4 2171.20  6003.6 2185.07  6041.2 2185.65
#Mann=7,-1,0
  2610.9   0.035       0  4942.6    0.07       0  4991.2    0.07       0
  5003.4    0.07       0  5211.5   0.035       0  5531.3    0.07       0
  6003.6   0.035       0
Bank Sta=4991.2,5003.4
Exp/Cntr=0.3,0.1

Type RM Length L Ch R = 1,30633,133,133,133
BEGIN DESCRIPTION:
Bull Creek 61.5
END DESCRIPTION:
XS GIS Cut Line= 4
      1328794.64      6920724.00      1329721.68      6920898.47
      1330131.65      6920917.96      1330705.80      6920093.42
#Sta/Elev= 30
  3699.8 2155.07  3852.2 2153.13  4234.7 2150.48  4449.7 2149.81  4473.5 2148.91
  4507.3 2149.73  4524.4 2148.93  4626.1 2148.75  4756.6 2146.68  4836.7 2143.86
  4926.8 2142.72  4956.8 2141.25  4976.8 2139.05  4986.8 2140.86  4996.8 2139.99
  5000.7 2132.99  5001.2 2132.49  5012.9 2132.99  5026.9 2139.20  5052.7 2142.96
  5063.9 2142.96  5070.0 2144.30  5089.6 2145.24  5135.4 2147.68  5377.7 2149.60
  5537.7 2153.16  5732.6 2159.59  5875.9 2164.49  5981.9 2168.96  6058.3 2170.66
#Mann=7,-1,0
  3699.8   0.035       0  5000.7   0.035       0  5012.9   0.035       0
  5089.6    0.07       0  5377.7   0.035       0  5732.6    0.07       0
  5875.9   0.035       0
Bank Sta=5000.7,5012.9
Exp/Cntr=0.3,0.1

Type RM Length L Ch R = 1,30500,500,500,500
BEGIN DESCRIPTION:
Bull Creek 61.0
END DESCRIPTION:
XS GIS Cut Line= 4
      1327667.52      6920478.75      1330004.18      6921020.78
      1330156.70      6921063.68      1330730.40      6920239.79
#Sta/Elev= 30
  2601.3 2178.85  2973.8 2164.79  3132.5 2160.04  3389.2 2157.54  3532.9 2157.47
  3543.1 2156.35  4005.1 2152.40  4508.1 2149.17  4571.1 2149.75  4580.0 2148.78
  4816.1 2146.42  4959.8 2142.31  4990.6 2139.69  5000.0 2136.55  5001.0 2131.38
  5001.5 2130.88  5013.2 2131.38  5021.6 2140.50  5032.0 2140.17  5063.2 2143.14
  5080.4 2142.74  5153.7 2145.82  5214.4 2146.15  5520.2 2147.58  5637.0 2149.22
  5735.1 2152.00  5909.9 2157.29  5960.4 2159.99  6094.6 2164.03  6162.4 2167.86
#Mann=9,-1,0
  2601.3   0.035       0  5001.0   0.035       0  5013.2   0.035       0
  5214.4    0.07       0  5520.2   0.035       0  5637.0    0.07       0
  5735.1   0.035       0  5909.9    0.07       0  5960.4   0.035       0
Bank Sta=5001,5013.2
Exp/Cntr=0.3,0.1

Type RM Length L Ch R = 1,30000,607,607,607
BEGIN DESCRIPTION:
Bull Creek 60.0
END DESCRIPTION:
XS GIS Cut Line= 4
      1327556.33      6920471.78      1330086.63      6921447.59
      1330163.13      6921394.25      1330955.02      6920387.98
#Sta/Elev= 30
  2194.8 2183.86  2725.1 2163.21  2839.6 2160.03  3450.8 2157.35  3644.5 2155.66
  3908.2 2150.81  4479.5 2147.74  4727.7 2146.49  4805.5 2143.65  4912.8 2144.60
  4948.6 2142.86  4954.7 2140.26  4969.5 2138.51  4977.9 2132.18  4978.3 2129.99
  4978.8 2129.49  4990.5 2129.99  4998.1 2136.86  5006.4 2137.96  5062.4 2137.74
  5097.7 2140.18  5262.5 2144.89  5372.9 2144.77  5375.7 2144.82  5724.8 2145.58
  5902.8 2148.72  6089.7 2155.74  6144.9 2158.59  6173.8 2162.17  6280.5 2169.46
#Mann=8,-1,0
  2194.8   0.035       0  4479.5    0.07       0  4805.5   0.035       0
  4978.3   0.035       0  4990.5   0.035       0  5372.9    0.07       0
  5375.7   0.035       0  6089.7    0.07       0
Bank Sta=4978.3,4990.5
Exp/Cntr=0.3,0.1

Type RM Length L Ch R = 1,29393,393,393,393
BEGIN DESCRIPTION:
Bull Creek 59.0
END DESCRIPTION:
XS GIS Cut Line= 4
      1330827.20      6923562.03      1330750.81      6921749.57
      1330674.42      6921464.85      1330954.99      6920438.05
#Sta/Elev= 30
  2885.3 2154.56  2915.4 2153.11  3013.5 2151.34  3089.5 2151.04  3139.6 2147.30
  3228.1 2146.25  3610.0 2144.84  3640.0 2145.85  3680.0 2144.32  4121.4 2142.12
  4239.6 2142.12  4340.6 2145.70  4420.7 2143.32  4590.8 2144.54  4854.0 2138.24
  4859.2 2139.47  4894.0 2140.02  4994.2 2134.41  5001.3 2132.23  5008.4 2126.72
  5008.9 2126.22  5023.8 2126.72  5032.4 2133.19  5063.5 2139.03  5104.9 2141.26
  5602.5 2142.63  5768.4 2147.03  5871.5 2153.07  5934.2 2155.77  6058.6 2164.15
#Mann=8,-1,0
  2885.3   0.035       0  2915.4    0.07       0  3013.5   0.035       0
  3228.1    0.07       0  4121.4   0.035       0  5008.4   0.035       0
  5023.8   0.035       0  5871.5    0.07       0
Bank Sta=5008.4,5023.8
Exp/Cntr=0.3,0.1

Type RM Length L Ch R = 1,29000,500,500,500
BEGIN DESCRIPTION:
Bull Creek 58.0
END DESCRIPTION:
XS GIS Cut Line= 3
      1330889.70      6923930.12      1331027.70      6921588.08
      1331014.70      6920332.95
#Sta/Elev= 30
  2653.9 2167.70  2672.7 2167.55  2856.4 2159.83  3050.3 2154.85  3148.2 2152.50
  3207.0 2152.27  3261.2 2148.57  3297.1 2149.33  3356.5 2146.43  3449.9 2145.17
  4332.1 2140.00  4649.5 2145.80  4769.4 2142.05  4781.8 2141.60  4960.0 2135.80
  4997.5 2128.03  5010.1 2129.62  5020.1 2127.59  5022.4 2124.80  5022.9 2124.30
  5037.8 2124.80  5040.1 2132.52  5090.1 2137.78  5150.1 2140.26  5680.1 2140.85
  5850.1 2146.23  6030.2 2156.57  6130.1 2163.20  6190.1 2176.89  6255.2 2177.81
#Mann=13,-1,0
  2653.9    0.07       0  2672.7   0.035       0  3050.3    0.07       0
  3148.2   0.035       0  3261.2    0.07       0  3356.5   0.035       0
  3449.9    0.07       0  4332.1   0.035       0  4769.4    0.07       0
  4781.8   0.035       0  5022.4   0.035       0  5037.8   0.035       0
  6030.2    0.07       0
Bank Sta=5022.4,5037.8
Exp/Cntr=0.3,0.1

Type RM Length L Ch R = 1,28500,500,500,500
BEGIN DESCRIPTION:
Bull Creek 57.0
END DESCRIPTION:
XS GIS Cut Line= 3
      1331505.00      6923237.96      1331402.30      6921340.34
      1331005.00      6920338.00
#Sta/Elev= 30
  3099.6 2151.84  3179.7 2147.91  3209.7 2148.66  3229.7 2146.49  3427.6 2142.62
  3571.2 2141.19  3733.0 2138.73  3884.5 2137.31  4177.3 2136.51  4532.7 2138.28
  4664.7 2138.32  4882.2 2136.48  4992.3 2132.24  5003.1 2131.47  5023.7 2123.70
  5024.2 2123.20  5039.1 2123.70  5045.5 2128.22  5061.1 2134.22  5090.8 2138.01
  5400.5 2139.00  5768.9 2151.16  5877.8 2158.07  5960.7 2165.25  5970.6 2167.81
  5979.6 2172.37  5985.0 2170.89  6009.3 2178.25  6014.7 2176.88  6078.2 2176.92
#Mann=11,-1,0
  3099.6    0.07       0  3427.6   0.035       0  3571.2    0.07       0
  3733.0   0.035       0  3884.5    0.07       0  4177.3   0.035       0
  4532.7    0.07       0  4664.7   0.035       0  5023.7   0.035       0
  5039.1   0.035       0  5877.8    0.07       0
Bank Sta=5023.7,5039.1
Exp/Cntr=0.3,0.1

Type RM Length L Ch R = 1,28000,500,500,500
BEGIN DESCRIPTION:
Bull Creek 56.0
END DESCRIPTION:
XS GIS Cut Line= 3
      1331504.99      6923188.04      1331833.68      6921288.26
      1331655.01      6920788.01
#Sta/Elev= 30
  3072.0 2149.22  3099.4 2147.91  3132.9 2148.72  3183.7 2145.68  3244.6 2145.80
  3264.9 2144.12  3328.0 2142.93  3366.3 2143.63  3386.6 2142.02  3496.5 2140.92
  3596.0 2139.71  3746.8 2137.31  3968.4 2136.05  4168.7 2135.76  4305.7 2136.43
  4786.0 2136.11  4929.2 2134.56  4959.7 2131.81  4969.8 2129.24  4976.7 2124.60
  4981.7 2127.29  4982.3 2120.48  4982.8 2119.98  4997.9 2120.48  5000.0 2124.79
  5002.8 2124.79  5008.3 2130.56  5064.0 2134.79  5233.9 2134.92  5531.2 2145.74
#Mann=10,-1,0
  3072.0    0.07       0  3328.0   0.035       0  3496.5    0.07       0
  3596.0   0.035       0  3968.4    0.07       0  4168.7   0.035       0
  4305.7    0.07       0  4786.0   0.035       0  4982.3   0.035       0
  4997.9   0.035       0
Bank Sta=4982.3,4997.9
Exp/Cntr=0.3,0.1

Type RM Length L Ch R = 1,27500,500,500,500
BEGIN DESCRIPTION:
Bull Creek 55.0
END DESCRIPTION:
XS GIS Cut Line= 3
      1331605.00      6923787.99      1332301.21      6921184.99
      1331955.00      6920687.99
#Sta/Elev= 30
  2305.5 2198.35  2357.2 2193.49  2419.4 2182.14  2471.1 2176.72  2523.2 2168.46
  2543.6 2170.15  2564.3 2165.78  2593.0 2163.10  2699.3 2158.71  2710.8 2158.71
  3081.9 2144.30  3402.1 2139.08  3733.0 2135.61  3836.4 2134.85  4086.8 2133.80
  4832.8 2133.58  4918.6 2132.62  4986.5 2128.73  4993.5 2123.83  5000.0 2126.67
  5000.7 2119.41  5001.2 2118.91  5016.3 2119.41  5017.1 2121.24  5023.2 2122.44
  5032.0 2130.04  5052.9 2131.66  5118.2 2130.90  5246.6 2137.10  5605.7 2147.96
#Mann=10,-1,0
  2305.5    0.07       0  2699.3   0.035       0  2710.8    0.07       0
  3402.1   0.035       0  3733.0    0.07       0  3836.4   0.035       0
  4086.8    0.07       0  4832.8   0.035       0  5000.7   0.035       0
  5016.3   0.035       0
Bank Sta=5000.7,5016.3
Exp/Cntr=0.3,0.1

Type RM Length L Ch R = 1,27000,500,500,500
BEGIN DESCRIPTION:
Bull Creek 54.0
END DESCRIPTION:
XS GIS Cut Line= 3
      1331773.40      6923221.10      1332778.27      6921160.68
      1332875.52      6920601.27
#Sta/Elev= 30
  2707.6 2151.15  2732.7 2150.24  2777.8 2147.38  2896.2 2144.31  2978.6 2143.73
  2995.6 2142.05  3130.8 2139.17  3215.0 2139.19  3294.1 2136.61  3467.6 2135.00
  4026.2 2134.40  4264.0 2130.71  4338.2 2132.04  4486.3 2132.48  4646.6 2132.22
  4849.0 2130.52  4868.9 2130.98  4983.7 2128.55  5003.9 2125.54  5006.2 2118.16
  5006.7 2117.66  5021.9 2118.16  5033.2 2120.09  5043.3 2126.07  5053.5 2129.09
  5068.6 2130.26  5083.9 2140.81  5104.2 2143.42  5256.5 2150.66  5567.8 2159.74
#Mann=12,-1,0
  2707.6    0.07       0  2732.7   0.035       0  2896.2    0.07       0
  3215.0   0.035       0  4264.0    0.07       0  4338.2   0.035       0
  4486.3    0.07       0  4646.6   0.035       0  4849.0    0.07       0
  4868.9   0.035       0  5006.2   0.035       0  5021.9   0.035       0
Bank Sta=5006.2,5021.9
Exp/Cntr=0.3,0.1

Type RM Length L Ch R = 1,26500,500,500,500
BEGIN DESCRIPTION:
Bull Creek 53.0
END DESCRIPTION:
XS GIS Cut Line= 3
      1331470.40      6923430.38      1333174.56      6921338.59
      1333043.35      6920576.20
#Sta/Elev= 30
  2301.9 2158.75  2605.1 2148.90  3154.4 2138.94  4020.8 2133.26  4226.6 2129.38
  4388.2 2131.46  4427.0 2131.36  4859.6 2130.56  4993.5 2126.50  5002.8 2123.96
  5013.0 2112.51  5013.5 2112.01  5028.7 2112.51  5041.2 2125.79  5051.3 2127.41
  5261.0 2130.95  5305.0 2134.54  5376.6 2147.46  5416.6 2160.09  5457.2 2181.26
  5477.5 2180.89  5495.6 2171.30  5500.7 2174.52  5518.1 2163.71  5538.4 2158.60
  5599.3 2154.86  5670.3 2165.90  5730.2 2185.42  5771.2 2183.09  5773.6 2183.09
#Mann=10,-1,0
  2301.9    0.07       0  3154.4   0.035       0  4020.8    0.07       0
  4388.2   0.035       0  4427.0    0.07       0  4859.6   0.035       0
  5013.0   0.035       0  5028.7   0.035       0  5376.6    0.07       0
  5771.2   0.035       0
Bank Sta=5013,5028.7
Exp/Cntr=0.3,0.1

Type RM Length L Ch R = 1,26000,500,500,500
BEGIN DESCRIPTION:
Bull Creek 52.0
END DESCRIPTION:
XS GIS Cut Line= 4
      1331449.57      6923305.37      1333543.34      6921154.30
      1333373.12      6920969.07      1333080.80      6920561.95
#Sta/Elev= 30
  1746.6 2153.25  2038.5 2145.58  2507.9 2138.98  2865.9 2134.40  3298.7 2133.30
  3601.3 2129.13  3749.9 2131.20  3902.8 2130.12  4275.8 2129.62  4718.7 2129.97
  4801.1 2128.95  4822.7 2126.24  4949.7 2126.27  4992.2 2124.36  4997.3 2118.38
  5002.7 2118.38  5005.8 2112.83  5006.3 2112.33  5021.5 2112.83  5042.0 2118.19
  5050.6 2123.58  5086.2 2126.61  5121.8 2134.22  5198.2 2138.10  5364.9 2147.66
  5400.6 2159.40  5436.2 2182.52  5465.6 2187.93  5498.4 2185.06  5501.2 2184.43
#Mann=10,-1,0
  1746.6    0.07       0  2507.9   0.035       0  3298.7    0.07       0
  3749.9   0.035       0  3902.8    0.07       0  4275.8   0.035       0
  5005.8   0.035       0  5021.5   0.035       0  5198.2    0.07       0
  5498.4   0.035       0
Bank Sta=5005.8,5021.5
Exp/Cntr=0.3,0.1

Type RM Length L Ch R = 1,25500,500,500,500
BEGIN DESCRIPTION:
Bull Creek 51.0
END DESCRIPTION:
XS GIS Cut Line= 3
      1331475.64      6923347.00      1333716.70      6921087.22
      1333631.89      6920128.26
#Sta/Elev= 30
  1817.4 2154.71  2134.4 2146.27  2613.9 2138.77  3390.3 2132.74  3683.0 2129.02
  3832.6 2130.81  3867.4 2130.84  3941.1 2130.32  4077.7 2129.66  4158.3 2128.67
  4220.5 2128.47  4391.2 2128.52  4643.8 2128.40  4695.2 2128.19  4920.5 2128.83
  4955.8 2121.84  4962.9 2123.30  4970.0 2116.16  4977.0 2118.16  4988.0 2109.76
  4988.5 2109.26  5003.8 2109.76  5029.3 2121.49  5075.3 2125.58  5089.6 2123.19
  5179.9 2128.27  5400.8 2130.93  5712.0 2144.02  5938.8 2146.17  5962.7 2146.42
#Mann=15,-1,0
  1817.4    0.07       0  2613.9   0.035       0  3390.3    0.07       0
  3832.6   0.035       0  3867.4    0.07       0  3941.1   0.035       0
  4077.7    0.07       0  4158.3   0.035       0  4220.5    0.07       0
  4391.2   0.035       0  4643.8    0.07       0  4695.2   0.035       0
  4988.0   0.035       0  5003.8   0.035       0  5938.8    0.07       0
Bank Sta=4988,5003.8
Exp/Cntr=0.3,0.1

Type RM Length L Ch R = 1,25000,500,500,500
BEGIN DESCRIPTION:
Bull Creek 50.0
END DESCRIPTION:
XS GIS Cut Line= 3
      1334080.67      6922196.81      1334178.94      6921188.38
      1333904.98      6920487.96
#Sta/Elev= 30
  3986.8 2142.63  4087.0 2142.81  4183.8 2138.66  4226.7 2139.27  4266.9 2135.01
  4323.8 2134.93  4457.8 2130.14  4804.6 2126.72  4829.6 2124.47  4839.6 2126.97
  4879.8 2125.03  4940.1 2126.88  4970.2 2118.92  4980.3 2111.99  4981.0 2107.07
  4981.5 2106.57  4999.6 2107.07  5000.0 2110.27  5002.9 2110.27  5011.2 2116.78
  5020.5 2120.71  5110.0 2125.12  5490.1 2126.11  5591.0 2127.90  5664.7 2131.87
  5676.9 2133.85  5707.3 2146.31  5730.6 2163.51  5737.1 2170.55  5752.1 2174.28
#Mann=5,-1,0
  3986.8    0.07       0  4323.8   0.035       0  4981.0   0.035       0
  4999.6   0.035       0  5664.7    0.07       0
Bank Sta=4981,4999.6
Exp/Cntr=0.3,0.1

Type RM Length L Ch R = 1,24500,97,97,97
BEGIN DESCRIPTION:
Bull Creek 49.0
END DESCRIPTION:
XS GIS Cut Line= 4
      1334445.25      6922623.89      1334372.34      6920868.71
      1334232.19      6920765.57      1333904.99      6920437.99
#Sta/Elev= 30
  3069.3 2140.61  3333.6 2136.25  3431.7 2135.24  3519.3 2134.76  3659.2 2133.98
  4246.2 2128.11  4286.2 2125.79  4306.3 2127.90  4477.0 2123.80  4616.5 2124.51
  4676.6 2129.51  4756.6 2122.67  4826.0 2121.57  4853.1 2118.64  4858.5 2115.51
  4859.0 2115.01  4877.1 2115.51  4888.6 2118.63  4917.9 2116.16  4924.1 2118.32
  4977.8 2118.14  5000.0 2117.76  5059.9 2125.63  5286.2 2128.31  5339.3 2133.83
  5349.9 2135.43  5385.2 2149.46  5406.4 2164.15  5434.7 2179.32  5463.0 2175.11
#Mann=10,-1,0
  3069.3   0.035       0  3333.6    0.07       0  3431.7   0.035       0
  3519.3    0.07       0  3659.2   0.035       0  4477.0    0.07       0
  4858.5   0.035       0  4877.1    0.07       0  4977.8   0.035       0
  5339.3    0.07       0
Bank Sta=4858.5,4877.1
Exp/Cntr=0.3,0.1

Type RM Length L Ch R = 1,24403,81,81,81
BEGIN DESCRIPTION:
Bull Creek 48.6
END DESCRIPTION:
XS GIS Cut Line= 4
      1334503.84      6922588.72      1334430.93      6920833.56
      1334290.78      6920730.41      1333963.64      6920402.89
#Sta/Elev= 30
  3013.6 2138.86  3155.7 2137.59  3235.9 2136.35  3531.9 2133.94  3535.4 2134.07
  4135.3 2128.44  4175.3 2126.10  4195.3 2129.17  4245.4 2125.97  4462.8 2123.86
  4595.7 2124.16  4655.7 2131.33  4821.5 2127.68  4907.1 2129.36  5011.5 2122.32
  5012.0 2121.82  5030.1 2122.32  5032.7 2122.48  5268.3 2128.45  5324.8 2134.31
  5346.1 2140.95  5353.1 2140.63  5360.2 2144.71  5367.3 2144.42  5374.3 2148.89
  5381.4 2146.73  5388.5 2152.02  5395.6 2148.26  5402.6 2152.12  5407.2 2147.68
#Mann=9,-1,0
  3013.6   0.035       0  3155.7    0.07       0  3235.9   0.035       0
  3531.9    0.07       0  3535.4   0.035       0  4462.8    0.07       0
  5011.5    0.07       0  5030.1    0.07       0  5032.7   0.035       0
Bank Sta=5011.5,5030.1
Exp/Cntr=0.3,0.1

Type RM Length L Ch R = 1,24322,322,322,322
BEGIN DESCRIPTION:
Bull Creek 48.5
END DESCRIPTION:
XS GIS Cut Line= 4
      1334503.85      6922476.78      1334494.36      6920787.13
      1334290.78      6920618.44      1333964.69      6920291.96
#Sta/Elev= 30
  3069.6 2138.49  3076.5 2138.84  3177.1 2136.26  3338.4 2134.14  3754.0 2132.43
  3808.4 2130.03  3998.4 2127.99  4038.4 2129.02  4108.4 2126.35  4128.4 2128.80
  4158.4 2126.78  4358.4 2123.22  4475.7 2123.85  4678.4 2123.59  4718.4 2125.63
  4745.9 2122.83  4784.1 2120.02  4819.9 2119.50  4820.4 2119.00  4838.5 2119.50
  4843.5 2121.16  4850.0 2120.61  4900.8 2124.64  4982.3 2124.95  5023.7 2121.78
  5084.6 2125.01  5148.3 2125.02  5190.7 2127.21  5261.4 2127.96  5485.1 2138.79
#Mann=9,-1,0
  3069.6   0.035       0  3076.5    0.07       0  3177.1   0.035       0
  4475.7    0.07       0  4745.9   0.035       0  4784.1    0.07       0
  4819.9   0.035       0  4838.5    0.07       0  4982.3   0.035       0
Bank Sta=4819.9,4838.5
Exp/Cntr=0.3,0.1

Type RM Length L Ch R = 1,24000,380,380,380
BEGIN DESCRIPTION:
Bull Creek 48.0
END DESCRIPTION:
XS GIS Cut Line= 4
      1334460.88      6922675.96      1334599.67      6920545.78
      1334502.17      6920464.21      1333918.78      6920433.88
#Sta/Elev= 30
  2865.3 2140.03  2933.4 2141.64  2963.5 2138.59  3164.7 2136.52  3179.4 2136.10
  4520.7 2123.32  4676.8 2123.24  4747.2 2124.59  4807.4 2118.27  4817.4 2108.99
  4818.1 2106.19  4818.6 2105.69  4836.8 2106.19  4837.4 2108.85  4846.8 2116.68
  4907.6 2124.25  4947.7 2123.56  4967.7 2111.70  4977.7 2110.50  5002.2 2115.40
  5008.5 2119.75  5065.7 2123.51  5414.7 2125.83  5564.9 2130.60  5604.9 2135.09
  5625.0 2140.63  5655.0 2155.57  5675.0 2171.19  5694.6 2176.07  5711.3 2175.72
#Mann=8,-1,0
  2865.3   0.035       0  3164.7    0.07       0  3179.4   0.035       0
  4520.7    0.07       0  4676.8   0.035       0  4818.1   0.035       0
  4836.8   0.035       0  5694.6    0.07       0
Bank Sta=4818.1,4836.8
Exp/Cntr=0.3,0.1

Type RM Length L Ch R = 1,23620,120,120,120
BEGIN DESCRIPTION:
Bull Creek 47.5
END DESCRIPTION:
XS GIS Cut Line= 3
      1334386.97      6921498.38      1334924.57      6920698.44
      1334586.95      6918698.44
#Sta/Elev= 30
  4025.9 2128.14  4082.8 2128.33  4118.8 2126.07  4139.9 2129.17  4154.8 2126.92
  4205.8 2125.73  4478.9 2122.99  4904.8 2122.34  4925.8 2120.57  4931.9 2121.53
  4940.8 2119.40  4976.8 2117.43  4982.9 2116.14  4987.0 2113.38  4992.5 2113.38
  4999.5 2107.17  5000.0 2106.67  5021.3 2107.17  5030.7 2114.29  5040.9 2117.39
  5076.8 2121.36  5132.1 2123.53  5178.1 2122.61  5274.6 2122.54  5688.2 2123.68
  6551.9 2126.88  6815.0 2125.59  6960.8 2132.14  6996.4 2135.48  7018.0 2135.65
#Mann=7,-1,0
  4025.9   0.035       0  4999.5   0.035       0  5021.3   0.035       0
  5178.1   0.045       0  5274.6    0.07       0  5688.2   0.045       0
  6960.8    0.07       0
Bank Sta=4999.5,5021.3
Exp/Cntr=0.3,0.1

Type RM Length L Ch R = 1,23500,190,190,190
BEGIN DESCRIPTION:
Bull Creek 47.0
END DESCRIPTION:
XS GIS Cut Line= 3
      1334505.03      6921487.96      1335042.62      6920688.02
      1334705.00      6918688.02
#Sta/Elev= 30
  4036.2 2128.37  4079.6 2126.63  4108.4 2128.60  4157.7 2128.48  4367.7 2124.03
  4698.8 2121.41  4928.7 2122.33  4943.7 2120.45  4958.6 2116.80  4973.6 2116.10
  4979.7 2117.31  4994.6 2108.73  5002.5 2108.33  5004.6 2105.81  5005.1 2105.31
  5026.4 2105.81  5030.4 2110.87  5040.6 2117.45  5050.7 2117.56  5070.9 2121.62
  5076.0 2119.75  5091.3 2122.53  5142.0 2122.84  5174.4 2121.48  6602.4 2126.14
  6795.1 2125.09  6866.5 2126.80  6957.3 2132.23  6967.5 2135.21  7028.3 2140.55
#Mann=5,-1,0
  4036.2   0.035       0  5004.6   0.035       0  5026.4   0.035       0
  5174.4   0.045       0  6866.5    0.07       0
Bank Sta=5004.6,5026.4
Exp/Cntr=0.3,0.1

Type RM Length L Ch R = 1,23310,127,127,127
BEGIN DESCRIPTION:
Bull Creek 46.5
END DESCRIPTION:
XS GIS Cut Line= 3
      1334706.36      6921470.67      1335244.01      6920670.66
      1334906.59      6918671.83
#Sta/Elev= 30
  4056.7 2125.75  4079.6 2127.07  4721.6 2120.36  4850.6 2121.89  4943.6 2121.16
  4958.6 2116.73  4979.6 2114.60  4983.7 2104.73  4984.2 2104.23  5005.5 2104.73
  5015.6 2104.88  5019.2 2108.56  5024.5 2108.56  5033.4 2115.74  5071.9 2119.17
  5102.1 2121.84  5134.8 2122.34  5152.4 2121.29  5171.6 2120.92  5283.4 2120.04
  5733.2 2121.34  5936.0 2124.12  5948.5 2123.28  6098.3 2122.83  6372.1 2125.02
  6867.3 2123.78  6899.5 2123.74  6919.7 2125.71  6960.3 2126.28  7047.7 2130.13
#Mann=7,-1,0
  4056.7   0.035       0  4983.7   0.035       0  5005.5   0.035       0
  5071.9    0.07       0  5152.4   0.035       0  5171.6   0.045       0
  6867.3   0.035       0
Bank Sta=4983.7,5005.5
Exp/Cntr=0.3,0.1

Type RM Length L Ch R = 1,23183,431,431,431
BEGIN DESCRIPTION:
Bull Creek 46.0
END DESCRIPTION:
XS GIS Cut Line= 4
      1334799.07      6921509.84      1335276.69      6920816.37
      1335403.65      6920653.61      1334782.92      6918235.98
#Sta/Elev= 30
  4045.8 2125.80  4698.7 2120.19  4806.2 2121.28  4871.8 2117.54  4936.1 2117.60
  4949.2 2116.31  4956.9 2113.44  4963.2 2115.18  4971.4 2110.36  4977.7 2114.20
  4985.8 2109.87  4992.2 2112.35  4999.9 2108.55  5016.5 2104.54  5017.0 2104.04
  5038.3 2104.54  5041.9 2115.17  5124.2 2121.34  5172.3 2123.18  5188.6 2120.44
  5226.0 2119.79  5502.7 2119.40  6518.0 2124.79  6956.5 2123.67  7159.7 2131.19
  7216.5 2135.81  7260.2 2137.26  7299.1 2139.48  7439.8 2141.41  7590.3 2150.11
#Mann=7,-1,0
  4045.8   0.035       0  5016.5   0.035       0  5038.3   0.035       0
  5124.2    0.07       0  5226.0   0.045       0  6956.5   0.035       0
  7260.2    0.07       0
Bank Sta=5016.5,5038.3
Exp/Cntr=0.3,0.1

Type RM Length L Ch R = 1,22752,453,453,453
BEGIN DESCRIPTION:
Bull Creek 45.5
END DESCRIPTION:
XS GIS Cut Line= 4
      1334549.05      6921850.14      1335458.77      6921117.51
      1335545.57      6921037.65      1335142.51      6919174.14
#Sta/Elev= 30
  3837.0 2132.99  4027.3 2132.36  4049.7 2130.24  4099.2 2129.94  4140.9 2127.49
  4291.2 2126.19  4347.2 2123.58  4369.6 2124.54  4419.2 2123.11  4895.9 2122.32
  4923.2 2120.69  4937.5 2117.08  4980.7 2112.70  4989.7 2102.93  4990.2 2102.43
  5011.6 2102.93  5016.0 2104.76  5023.4 2112.64  5080.1 2119.76  5340.6 2121.55
  5543.9 2120.86  5593.3 2122.68  5603.5 2119.99  5644.7 2119.52  6084.4 2119.48
  6333.5 2121.65  6613.5 2121.57  6800.2 2122.77  6821.0 2124.25  7029.6 2123.52
#Mann=5,-1,0
  3837.0   0.035       0  4989.7   0.035       0  5011.6   0.035       0
  5543.9    0.07       0  5644.7   0.045       0
Bank Sta=4989.7,5011.6
Exp/Cntr=0.3,0.1

Type RM Length L Ch R = 1,22299,299,299,299
BEGIN DESCRIPTION:
Bull Creek 45.0
END DESCRIPTION:
XS GIS Cut Line= 4
      1336342.57      6921939.34      1335840.83      6921374.41
      1335590.22      6920879.24      1334887.09      6918183.89
#Sta/Elev= 30
  4117.2 2151.56  4150.5 2151.78  4201.1 2150.28  4208.7 2147.75  4286.4 2143.65
  4470.4 2135.53  4941.3 2118.73  4958.0 2117.37  4963.6 2114.85  4969.6 2106.19
  4980.8 2102.06  4981.3 2101.56  5003.2 2102.06  5024.8 2109.32  5030.4 2113.20
  5141.8 2114.55  5180.8 2119.11  5687.2 2120.89  5728.7 2122.44  5744.9 2119.35
  5789.2 2119.17  6811.9 2121.47  7009.2 2124.18  7314.0 2123.60  7397.8 2122.98
  7521.6 2122.26  7661.3 2124.52  7857.7 2131.01  8040.9 2139.23  8213.3 2149.56
#Mann=9,-1,0
  4117.2    0.07       0  4150.5   0.035       0  4980.8   0.035       0
  5003.2   0.035       0  5687.2    0.07       0  5789.2   0.045       0
  7314.0   0.035       0  7397.8   0.045       0  7521.6   0.035       0
Bank Sta=4980.8,5003.2
Exp/Cntr=0.3,0.1

Type RM Length L Ch R = 1,22000,500,500,500
BEGIN DESCRIPTION:
Bull Creek 44.0
END DESCRIPTION:
XS GIS Cut Line= 4
      1336306.35      6921543.28      1335905.43      6921005.85
      1335731.70      6920829.09      1334835.02      6918157.92
#Sta/Elev= 30
  4329.5 2139.59  4485.1 2133.83  4512.2 2130.94  4641.5 2125.50  4934.9 2117.71
  4977.1 2112.44  4984.8 2107.63  4985.0 2099.99  4985.5 2099.49  5007.4 2099.99
  5012.9 2100.13  5020.0 2103.19  5027.0 2111.19  5076.6 2113.41  5111.9 2118.27
  5455.7 2120.15  5491.6 2122.55  5512.7 2118.75  5559.9 2118.42  5884.4 2118.38
  7117.7 2123.62  7209.6 2122.92  7331.9 2122.25  7392.8 2124.36  7474.7 2124.52
  7717.3 2133.45  7886.1 2141.72  7897.3 2143.56  8008.0 2149.67  8065.5 2153.60
#Mann=9,-1,0
  4329.5   0.035       0  4985.0   0.035       0  5007.4   0.035       0
  5455.7    0.07       0  5559.9   0.045       0  7117.7   0.035       0
  7209.6   0.045       0  7331.9   0.035       0  8008.0    0.07       0
Bank Sta=4985,5007.4
Exp/Cntr=0.3,0.1

Type RM Length L Ch R = 1,21500,500,500,500
BEGIN DESCRIPTION:
Bull Creek 43.0
END DESCRIPTION:
XS GIS Cut Line= 3
      1336354.99      6921387.96      1336130.35      6920612.12
      1334959.56      6918247.16
#Sta/Elev= 30
  4192.3 2134.71  4473.3 2123.44  4733.6 2118.93  4796.1 2113.19  4894.2 2112.85
  4927.8 2110.91  4941.8 2108.25  4955.4 2102.25  4955.9 2101.75  4977.8 2102.25
  4999.5 2102.48  5022.3 2116.69  5064.8 2116.88  5072.8 2116.61  5089.6 2108.44
  5105.0 2105.56  5112.0 2110.28  5117.6 2107.79  5127.3 2115.57  5155.5 2114.80
  5246.6 2112.53  5252.2 2114.37  5313.9 2116.25  5633.5 2116.49  5796.8 2119.62
  5874.6 2118.20  6933.3 2121.29  7292.1 2126.91  7455.7 2132.88  7638.9 2143.69
#Mann=6,-1,0
  4192.3   0.035       0  4955.4   0.035       0  4977.8   0.035       0
  5064.8    0.07       0  5155.5   0.045       0  6933.3   0.035       0
Bank Sta=4955.4,4977.8
Exp/Cntr=0.3,0.1

Type RM Length L Ch R = 1,21000,500,500,500
BEGIN DESCRIPTION:
Bull Creek 42.0
END DESCRIPTION:
XS GIS Cut Line= 3
      1336527.72      6921634.49      1336528.66      6920715.99
      1335043.34      6918118.82
#Sta/Elev= 30
  4081.5 2136.56  4388.0 2129.11  4577.6 2122.39  4650.3 2120.35  4798.0 2117.59
  4918.0 2111.69  4948.0 2112.93  4959.0 2105.38  4966.8 2099.77  4967.3 2099.27
  4989.2 2099.77  5030.2 2101.88  5070.1 2103.40  5089.8 2105.03  5096.8 2109.85
  5102.6 2106.04  5112.6 2111.50  5118.4 2108.53  5124.4 2111.70  5140.0 2114.88
  5161.2 2116.16  5321.3 2113.89  5815.6 2114.85  5887.0 2116.93  6679.6 2117.06
  7260.5 2120.47  7697.8 2131.05  7896.4 2139.14  7939.6 2139.11  7991.9 2143.12
#Mann=11,-1,0
  4081.5   0.035       0  4577.6    0.07       0  4650.3   0.035       0
  4959.0    0.07       0  4966.8    0.07       0  4989.2    0.07       0
  5030.2   0.035       0  5070.1   0.045       0  5161.2    0.07       0
  5321.3   0.045       0  7260.5   0.035       0
Bank Sta=4966.8,4989.2
Exp/Cntr=0.3,0.1

Type RM Length L Ch R = 1,20500,500,500,500
BEGIN DESCRIPTION:
Bull Creek 41.0
END DESCRIPTION:
XS GIS Cut Line= 5
      1337369.76      6921300.28      1336695.00      6920295.46
      1336604.92      6920240.66      1336497.08      6920163.52
      1335043.32      6918249.00
#Sta/Elev= 30
  3684.2 2138.43  3850.1 2136.01  3994.6 2132.68  4445.8 2115.84  4601.7 2114.25
  4632.7 2114.13  4776.5 2114.48  4885.5 2114.25  4958.0 2108.40  4973.5 2099.95
  4976.9 2094.67  4977.4 2094.17  4999.4 2094.67  5000.0 2097.34  5003.0 2097.34
  5009.6 2106.60  5021.6 2106.99  5024.3 2107.53  5030.5 2102.47  5045.2 2101.44
  5060.0 2105.97  5066.1 2110.85  5087.0 2114.21  5159.9 2113.29  5538.1 2114.36
  5666.9 2117.10  6465.7 2117.18  6929.0 2120.31  7328.8 2129.52  7536.5 2139.16
#Mann=11,-1,0
  3684.2   0.035       0  3850.1    0.07       0  3994.6   0.035       0
  4601.7    0.07       0  4632.7   0.035       0  4776.5   0.045       0
  4976.9   0.045       0  4999.4   0.045       0  5021.6    0.07       0
  5159.9   0.045       0  6929.0   0.035       0
Bank Sta=4976.9,4999.4
Exp/Cntr=0.3,0.1

Type RM Length L Ch R = 1,20000,379,379,379
BEGIN DESCRIPTION:
Bull Creek 40.0
END DESCRIPTION:
XS GIS Cut Line= 5
      1337425.29      6921230.79      1336875.55      6920260.74
      1336911.15      6920194.60      1336938.05      6920104.49
      1335205.01      6918188.01
#Sta/Elev= 30
  3809.9 2140.28  3857.3 2143.00  4051.5 2140.51  4077.5 2139.87  4127.0 2133.79
  4326.1 2126.71  4509.4 2116.41  4649.3 2111.96  4794.9 2113.54  4919.1 2112.73
  4955.9 2109.42  4973.1 2103.15  4982.8 2095.18  4983.3 2094.68  5005.3 2095.18
  5006.9 2098.03  5017.3 2101.15  5032.0 2109.15  5065.1 2116.56  5089.6 2113.46
  5138.5 2112.96  6191.3 2114.48  6531.3 2117.37  6558.9 2116.04  6898.9 2118.63
  6976.8 2121.48  7061.8 2121.07  7293.2 2126.04  7501.2 2131.91  7677.9 2139.74
#Mann=8,-1,0
  3809.9   0.035       0  4051.5    0.07       0  4794.9   0.035       0
  4973.1    0.07       0  4982.8    0.07       0  5005.3    0.07       0
  5138.5   0.045       0  7293.2   0.035       0
Bank Sta=4982.8,5005.3
Exp/Cntr=0.3,0.1

Type RM Length L Ch R = 1,19621,304,304,304
BEGIN DESCRIPTION:
Bull Creek 39.5
END DESCRIPTION:
XS GIS Cut Line= 5
      1337424.51      6921201.26      1337255.45      6920381.35
      1337253.46      6920304.48      1337280.37      6920214.37
      1335547.30      6918297.86
#Sta/Elev= 30
  4068.7 2141.70  4139.5 2143.63  4234.9 2141.27  4285.2 2135.23  4481.7 2126.87
  4707.1 2116.56  4872.0 2110.71  4939.2 2111.45  4949.2 2105.98  4978.3 2095.09
  4978.8 2094.59  5000.8 2095.09  5038.5 2099.64  5043.7 2098.41  5071.7 2104.54
  5085.4 2105.93  5106.4 2113.10  5127.3 2111.88  5288.0 2111.51  6756.3 2115.24
  6805.6 2117.45  6840.7 2116.13  7081.4 2118.58  7145.6 2121.79  7194.9 2120.70
  7237.5 2122.96  7449.7 2124.85  7506.5 2127.48  7570.0 2127.46  7660.7 2130.42
#Mann=7,-1,0
  4068.7   0.035       0  4481.7    0.07       0  4707.1   0.035       0
  4872.0    0.07       0  4978.3    0.07       0  5000.8    0.07       0
  5288.0   0.045       0
Bank Sta=4978.3,5000.8
Exp/Cntr=0.3,0.1

Type RM Length L Ch R = 1,19317,360,360,360
BEGIN DESCRIPTION:
Bull Creek 39.0
END DESCRIPTION:
XS GIS Cut Line= 5
      1337439.17      6921230.85      1337536.40      6920362.74
      1337677.64      6920041.99      1337879.03      6919101.02
      1337154.97      6918287.97
#Sta/Elev= 30
  4132.3 2139.64  4235.8 2138.49  4296.2 2141.92  4320.4 2139.28  4326.4 2141.27
  4376.7 2134.67  4447.1 2130.67  4940.2 2111.61  4951.8 2110.71  4994.4 2094.38
  4994.9 2093.88  5017.1 2094.38  5032.9 2098.17  5039.0 2102.42  5062.3 2106.05
  5109.0 2105.88  5114.4 2101.92  5166.6 2098.81  5295.1 2106.00  5327.9 2110.95
  5902.4 2111.19  5944.7 2109.29  6096.7 2111.67  6373.4 2110.04  6528.8 2111.75
  6560.3 2111.87  7059.9 2121.95  7095.8 2124.80  7396.7 2127.55  7407.3 2127.69
#Mann=6,-1,0
  4132.3   0.035       0  4994.4   0.035       0  5017.1   0.035       0
  6528.8   0.045       0  6560.3    0.07       0  7396.7   0.035       0
Bank Sta=4994.4,5017.1
Exp/Cntr=0.3,0.1

Type RM Length L Ch R = 1,18957,457,457,457
BEGIN DESCRIPTION:
Bull Creek 38.0
END DESCRIPTION:
XS GIS Cut Line= 6
      1337522.49      6921258.62      1337858.19      6920329.38
      1337859.93      6920200.32      1337983.19      6919573.59
      1338146.39      6918829.38      1338371.21      6917793.73
#Sta/Elev= 30
  3973.7 2146.55  4146.4 2142.30  4263.5 2133.80  4345.1 2128.58  4601.7 2118.67
  4654.8 2119.06  4708.0 2114.53  4785.4 2112.83  4881.1 2108.80  4941.2 2097.60
  4941.7 2097.10  4963.9 2097.60  5013.1 2100.22  5054.3 2108.20  5083.1 2111.41
  5141.0 2106.92  5184.9 2106.18  5205.3 2108.99  5243.8 2110.23  5403.0 2108.89
  5745.5 2110.21  5810.0 2108.27  5888.8 2110.70  6088.3 2109.85  7121.7 2115.55
  7165.7 2114.15  7342.2 2116.68  7383.1 2114.66  7455.5 2118.33  7551.2 2119.40
#Mann=6,-1,0
  3973.7    0.07       0  4263.5   0.045       0  4785.4    0.07       0
  4941.2    0.07       0  4963.9    0.07       0  5054.3   0.045       0
Bank Sta=4941.2,4963.9
Exp/Cntr=0.3,0.1

Type RM Length L Ch R = 1,18500,500,500,500
BEGIN DESCRIPTION:
Bull Creek 37.0
END DESCRIPTION:
XS GIS Cut Line= 4
      1338155.00      6920788.00      1338262.71      6920138.06
      1338281.55      6920037.18      1338503.74      6918058.34
#Sta/Elev= 30
  4341.2 2129.48  4418.5 2120.75  4594.6 2111.07  4706.1 2110.21  4740.2 2107.85
  4856.1 2107.96  4949.4 2104.65  4984.1 2100.05  4986.0 2095.00  4986.5 2094.50
  5009.0 2095.00  5020.4 2095.98  5037.7 2102.90  5062.5 2104.61  5132.0 2107.12
  5413.7 2106.21  5454.0 2103.55  5554.6 2102.44  5584.8 2104.64  5615.0 2103.70
  5816.3 2108.27  6344.0 2108.96  6429.0 2111.23  6460.3 2109.83  6742.0 2111.14
  6802.4 2113.34  6842.7 2111.70  6933.2 2114.61  6974.6 2113.40  7093.9 2115.21
#Mann=6,-1,0
  4341.2    0.07       0  4418.5   0.045       0  4856.1    0.07       0
  4986.0    0.07       0  5009.0    0.07       0  5062.5   0.045       0
Bank Sta=4986,5009
Exp/Cntr=0.3,0.1

Type RM Length L Ch R = 1,18000,500,500,500
BEGIN DESCRIPTION:
Bull Creek 36.0
END DESCRIPTION:
XS GIS Cut Line= 5
      1338184.58      6920785.05      1338635.97      6920271.16
      1338730.32      6920138.23      1338707.64      6920050.01
      1338594.88      6918253.63
#Sta/Elev= 30
  4153.0 2128.60  4194.7 2123.63  4391.9 2110.84  4477.3 2110.37  4561.8 2107.20
  4853.1 2106.68  4928.0 2101.10  4952.5 2099.51  4961.1 2097.01  4967.3 2097.90
  4975.8 2093.17  4976.7 2091.08  4977.2 2090.58  4999.7 2091.08  5010.6 2094.60
  5020.9 2102.02  5031.2 2103.94  5159.0 2105.84  5493.9 2105.87  5634.2 2100.30
  5724.3 2102.87  5754.4 2105.62  5924.7 2105.12  6275.4 2109.25  6395.7 2108.25
  6485.4 2109.14  6505.9 2111.03  6706.3 2110.42  6826.5 2113.20  6891.0 2112.08
#Mann=6,-1,0
  4153.0    0.07       0  4194.7   0.045       0  4928.0    0.07       0
  4976.7    0.07       0  4999.7    0.07       0  5159.0   0.045       0
Bank Sta=4976.7,4999.7
Exp/Cntr=0.3,0.1

Type RM Length L Ch R = 1,17500,500,500,500
BEGIN DESCRIPTION:
Bull Creek 35.0
END DESCRIPTION:
XS GIS Cut Line= 4
      1338800.36      6920302.64      1339137.13      6919960.65
      1339136.41      6919906.53      1338994.21      6918162.81
#Sta/Elev= 30
  4465.9 2105.57  4677.9 2105.54  4939.1 2103.32  4978.5 2100.51  4996.8 2093.16
  5017.1 2090.17  5017.6 2089.67  5040.1 2090.17  5048.7 2092.57  5058.7 2100.80
  5068.8 2103.32  5106.4 2103.74  5369.7 2102.94  5399.8 2104.13  5446.5 2100.75
  5520.2 2098.85  5560.4 2101.16  5590.5 2100.50  5781.1 2105.18  5811.2 2103.89
  6252.7 2105.55  6308.5 2108.07  6403.2 2108.02  6430.2 2110.53  6543.6 2110.26
  6583.8 2112.75  6623.9 2111.26  6664.0 2114.44  6704.2 2113.03  6749.5 2115.24
#Mann=5,-1,0
  4465.9   0.045       0  4677.9    0.07       0  5017.1    0.07       0
  5040.1    0.07       0  5106.4   0.045       0
Bank Sta=5017.1,5040.1
Exp/Cntr=0.3,0.1

Type RM Length L Ch R = 1,17000,127,127,127
BEGIN DESCRIPTION:
Bull Creek 34.0
END DESCRIPTION:
XS GIS Cut Line= 4
      1338819.85      6920295.73      1339191.97      6919933.52
      1339557.81      6919784.55      1339311.03      6918175.57
#Sta/Elev= 30
  4085.7 2105.70  4277.3 2104.89  4314.1 2106.89  4328.2 2102.59  4335.2 2105.29
  4342.4 2102.57  4349.4 2105.53  4356.5 2101.26  4363.5 2104.99  4391.8 2104.90
  4399.0 2100.70  4420.1 2102.95  4441.4 2099.65  4448.4 2102.65  4539.2 2103.60
  4979.2 2097.95  5000.0 2095.54  5015.4 2087.85  5015.9 2087.35  5038.4 2087.85
  5077.4 2091.81  5097.7 2102.24  5184.7 2101.87  5383.7 2096.90  5461.9 2100.12
  5593.4 2099.03  5647.1 2102.61  5785.6 2104.52  6048.7 2104.75  6627.8 2118.90
#Mann=6,-1,0
  4085.7   0.045       0  4277.3    0.07       0  4539.2   0.045       0
  5015.4   0.045       0  5038.4   0.045       0  5184.7   0.045       0
Bank Sta=5015.4,5038.4
Exp/Cntr=0.3,0.1

Type RM Length L Ch R = 1,16873,108,108,108
BEGIN DESCRIPTION:
Bull Creek 33.6
END DESCRIPTION:
XS GIS Cut Line= 4
      1338831.77      6920286.14      1339232.12      6919923.75
      1339736.38      6919794.48      1339758.08      6918336.11
#Sta/Elev= 30
  3999.9 2105.52  4175.5 2104.19  4213.3 2106.89  4234.2 2102.12  4241.7 2104.05
  4255.8 2098.76  4270.0 2100.46  4276.8 2105.03  4298.4 2104.68  4305.2 2100.19
  4312.6 2103.71  4319.4 2099.73  4341.0 2097.48  4359.4 2100.90  4524.8 2104.45
  4899.8 2098.15  4943.0 2097.19  4955.8 2090.66  4972.3 2087.85  4972.8 2087.35
  4995.3 2087.85  4997.1 2093.98  5005.5 2098.04  5017.8 2102.72  5527.0 2096.81
  5677.0 2102.78  5707.0 2100.92  5817.0 2104.31  5857.0 2102.70  6519.0 2119.69
#Mann=7,-1,0
  3999.9   0.045       0  4175.5    0.07       0  4359.4   0.045       0
  4899.8    0.07       0  4972.3    0.07       0  4995.3    0.07       0
  5005.5   0.045       0
Bank Sta=4972.3,4995.3
Exp/Cntr=0.3,0.1

Type RM Length L Ch R = 1,16765,765,765,765
BEGIN DESCRIPTION:
Bull Creek 33.5a
END DESCRIPTION:
XS GIS Cut Line= 5
      1338839.63      6920281.28      1339244.05      6919929.18
      1339271.29      6919919.20      1339775.44      6919907.32
      1340096.62      6918475.01
#Sta/Elev= 30
  4000.5 2105.62  4166.6 2103.91  4205.5 2106.68  4226.4 2102.12  4233.0 2104.05
  4254.8 2096.58  4269.1 2105.20  4315.8 2101.27  4332.7 2095.81  4339.3 2100.45
  4346.9 2098.74  4353.6 2100.73  4510.2 2104.45  4852.5 2099.58  4959.5 2097.62
  4979.6 2093.83  4988.1 2088.09  4988.6 2087.59  5011.1 2088.09  5039.6 2093.77
  5059.6 2102.36  5113.6 2101.86  5460.2 2100.14  5590.2 2095.66  5714.6 2098.05
  5881.3 2100.39  5940.4 2103.69  6124.9 2104.58  6247.9 2110.23  6537.9 2116.26
#Mann=9,-1,0
  4000.5   0.045       0  4166.6    0.07       0  4315.8   0.045       0
  4852.5    0.07       0  4988.1    0.07       0  5011.1    0.07       0
  5113.6   0.045       0  5714.6   0.035       0  5881.3   0.045       0
Bank Sta=4988.1,5011.1
Exp/Cntr=0.3,0.1

Type RM Length L Ch R = 1,16000,1000,1000,1000
BEGIN DESCRIPTION:
Bull Creek 32.0
END DESCRIPTION:
XS GIS Cut Line= 4
      1338155.00      6920838.00      1339158.34      6920186.31
      1339740.72      6920267.57      1340270.11      6918557.88
#Sta/Elev= 30
  3803.6 2131.99  3832.3 2131.98  3891.9 2125.30  4113.6 2111.41  4215.8 2108.22
  4854.4 2104.01  4880.2 2102.83  4895.3 2098.28  4901.3 2101.55  4952.6 2097.99
  4983.5 2088.47  4984.0 2087.97  5006.6 2088.47  5016.8 2089.32  5045.2 2099.35
  5050.3 2097.51  5077.4 2104.04  5119.7 2104.31  5226.1 2104.22  5349.9 2104.14
  6372.7 2099.86  6540.2 2095.54  6843.8 2103.16  6973.2 2103.12  7063.6 2108.05
  7095.0 2105.97  7126.4 2109.99  7271.9 2114.44  7304.4 2111.77  7377.8 2113.60
#Mann=8,-1,0
  3803.6    0.07       0  3891.9   0.045       0  4854.4    0.07       0
  4983.5    0.07       0  5006.6    0.07       0  5119.7   0.045       0
  5226.1    0.07       0  5349.9   0.045       0
Bank Sta=4983.5,5006.6
Exp/Cntr=0.3,0.1

Type RM Length L Ch R = 1,15000,500,500,500
BEGIN DESCRIPTION:
Bull Creek 30.0
END DESCRIPTION:
XS GIS Cut Line= 3
      1339404.98      6921238.04      1339804.22      6920433.34
      1340370.04      6918648.69
#Sta/Elev= 30
  4101.7 2105.96  4726.6 2101.40  4877.8 2101.20  4922.6 2095.64  4928.2 2098.13
  4939.0 2097.93  4945.0 2093.90  4950.6 2095.33  4967.4 2088.85  4973.0 2089.82
  5003.4 2085.51  5003.9 2085.01  5026.6 2085.51  5052.5 2090.32  5058.1 2093.57
  5084.8 2099.78  5100.0 2101.68  5133.2 2101.05  5698.0 2100.91  5970.7 2099.24
  6128.1 2095.06  6264.5 2100.04  6509.5 2102.40  6579.3 2107.51  6611.6 2104.93
  6670.9 2111.91  6708.5 2109.41  6773.0 2114.53  6810.6 2110.75  6872.2 2111.71
#Mann=5,-1,0
  4101.7   0.045       0  4726.6    0.07       0  5003.4    0.07       0
  5026.6    0.07       0  5133.2   0.045       0
Bank Sta=5003.4,5026.6
Exp/Cntr=0.3,0.1

Type RM Length L Ch R = 1,14500,500,500,500
BEGIN DESCRIPTION:
Bull Creek 29.0
END DESCRIPTION:
XS GIS Cut Line= 4
      1339771.21      6921650.28      1340240.59      6920388.66
      1340234.15      6920316.15      1340417.80      6918713.74
#Sta/Elev= 30
  3653.9 2108.69  3901.7 2103.60  4584.7 2099.73  4791.3 2099.55  4845.8 2099.18
  4872.7 2098.98  4911.1 2093.45  4966.5 2090.04  4967.8 2085.67  4968.3 2085.17
  4991.0 2085.67  5020.7 2087.50  5030.8 2095.58  5050.9 2099.18  5121.5 2099.13
  5566.3 2100.20  5805.7 2097.36  5823.8 2099.20  5866.1 2096.06  6017.1 2094.90
  6107.7 2096.24  6147.9 2099.28  6339.2 2100.94  6399.6 2103.05  6429.8 2107.02
  6460.0 2104.45  6527.4 2111.23  6560.6 2111.16  6590.8 2114.04  6685.7 2110.63
#Mann=7,-1,0
  3653.9   0.045       0  4584.7    0.07       0  4791.3   0.045       0
  4845.8    0.07       0  4967.8    0.07       0  4991.0    0.07       0
  5121.5   0.045       0
Bank Sta=4967.8,4991
Exp/Cntr=0.3,0.1

Type RM Length L Ch R = 1,14000,500,500,500
BEGIN DESCRIPTION:
Bull Creek 28.0
END DESCRIPTION:
XS GIS Cut Line= 3
      1341239.94      6921228.36      1340691.84      6920437.90
      1340612.24      6920033.05
#Sta/Elev= 30
  4038.1 2112.30  4172.4 2114.21  4250.0 2112.93  4294.1 2113.71  4379.3 2106.57
  4397.0 2106.54  4488.5 2105.67  4512.0 2104.24  4560.1 2101.20  4724.3 2099.83
  4804.6 2097.20  4861.4 2092.19  4939.1 2090.36  4947.8 2089.02  4962.7 2084.51
  4963.4 2083.22  4963.9 2082.72  4987.6 2083.22  5012.4 2084.75  5020.3 2089.67
  5050.9 2091.72  5058.7 2095.02  5063.8 2093.80  5071.2 2096.97  5110.1 2100.47
  5122.2 2099.00  5166.5 2098.50  5275.1 2099.78  5315.6 2098.13  5412.6 2098.20
#Mann=5,-1,0
  4038.1   0.045       0  4397.0   0.035       0  4512.0    0.07       0
  4963.4    0.07       0  4987.6    0.07       0
Bank Sta=4963.4,4987.6
Exp/Cntr=0.3,0.1

Type RM Length L Ch R = 1,13500,500,500,500
BEGIN DESCRIPTION:
Bull Creek 27.0
END DESCRIPTION:
XS GIS Cut Line= 3
      1341205.00      6920938.01      1341139.04      6920287.95
      1340684.19      6919989.73
#Sta/Elev= 30
  4346.6 2113.62  4372.9 2111.61  4394.0 2108.60  4437.1 2107.19  4457.2 2105.36
  4477.3 2105.51  4516.9 2103.63  4587.8 2100.69  4768.8 2097.94  4809.0 2098.55
  4859.2 2094.46  4892.9 2096.47  4929.6 2092.97  4949.7 2088.59  4969.8 2087.49
  4979.8 2084.23  4985.3 2080.27  4985.8 2079.77  5009.6 2080.27  5025.0 2081.00
  5031.0 2082.54  5040.1 2083.18  5046.1 2088.15  5061.2 2087.81  5067.2 2090.43
  5088.5 2096.31  5103.3 2098.15  5432.9 2097.54  5543.4 2097.81  5543.9 2097.81
#Mann=7,-1,0
  4346.6   0.045       0  4372.9   0.035       0  4516.9    0.07       0
  4985.3    0.07       0  5009.6    0.07       0  5432.9   0.045       0
  5543.4    0.07       0
Bank Sta=4985.3,5009.6
Exp/Cntr=0.3,0.1
