--- Cottonwood Creek Trib034.prj (project) ---

Proj Title=Cottonwood Creek Trib034 Base Level Engineering
Current Plan=p01
Default Exp/Contr=0.3,0.1
English Units
Geom File=g01
Flow File=f01
Plan File=p01
BEGIN DESCRIPTION:
Cottonwood Creek Trib034
END DESCRIPTION:

--- Cottonwood Creek Trib034.p01 (plan) ---

Plan Title=Multiple Run
Short Identifier=Multiple
Geom File=g01
Flow File=f01
Subcritical Flow
K Sum by GR= 0
Std Step Tol= 0.01
Critical Tol= 0.01
Num of Std Step Trials= 20
Max Error Tol= 0.3
Flow Tol Ratio= 0.001
Split Flow NTrial= 30
Split Flow Tol= 0.02
Split Flow Ratio= 0.02
Log Output Level= 0
Friction Slope Method= 1
Unsteady Friction Slope Method= 2
Unsteady Bridges Friction Slope Method= 1
Parabolic Critical Depth
Global Vel Dist=  1 , 1 , 1
Global Log Level= 0
CheckData=True
Encroach Param= -1, 0, 0, 0
BEGIN DESCRIPTION:
Multiple Run
END DESCRIPTION:

--- Cottonwood Creek Trib034.f01 (steady flow) ---

Flow Title=Multiple
Number of Profiles=7
Profile Names=10-year,25-year,50-year,1pct_min,100-year,1pct_plu,500-year
River Rch & RM= Cottonwood Creek,Reach-1,36179
     197     271     331     201     401     801     597
River Rch & RM= Cottonwood Creek,Reach-1,33500
     273     381     469     287     573    1143     864
River Rch & RM= Cottonwood Creek,Reach-1,27500
     310     435     538     330     658    1312     999
River Rch & RM= Cottonwood Creek,Reach-1,26000
     383     541     673     414     827    1650    1267
River Rch & RM= Cottonwood Creek,Reach-1,22500
     620     894    1126     701    1399    2791    2193
River Rch & RM= Cottonwood Creek,Reach-1,15500
     723    1045    1319     823    1642    3275    2582
River Rch & RM= Cottonwood Creek,Reach-1,11000
     741    1070    1349     840    1676    3345    2629
River Rch & RM= Cottonwood Creek,Reach-1,7500
     774    1120    1413     881    1758    3507    2762
River Rch & RM= Cottonwood Creek,Reach-1,6500
     805    1166    1472     918    1832    3655    2881
River Rch & RM= Cottonwood Creek,Reach-1,5500
     842    1221    1543     964    1923    3836    3028
River Rch & RM= Cottonwood Creek,Reach-1,5000
     897    1305    1653    1034    2063    4115    3262
River Rch & RM= Cottonwood Creek,Reach-1,2500
     940    1371    1740    1091    2177    4343    3456
Boundary for River Rch & Prof#=Cottonwood Creek,Reach-1,1
Up Type=0
Dn Type=3
Dn Slope=0.005
Boundary for River Rch & Prof#=Cottonwood Creek,Reach-1,2
Up Type=0
Dn Type=3
Dn Slope=0.005
Boundary for River Rch & Prof#=Cottonwood Creek,Reach-1,3
Up Type=0
Dn Type=3
Dn Slope=0.005
Boundary for River Rch & Prof#=Cottonwood Creek,Reach-1,4
Up Type=0
Dn Type=3
Dn Slope=0.005
Boundary for River Rch & Prof#=Cottonwood Creek,Reach-1,5
Up Type=0
Dn Type=3
Dn Slope=0.005
Boundary for River Rch & Prof#=Cottonwood Creek,Reach-1,6
Up Type=0
Dn Type=3
Dn Slope=0.005
Boundary for River Rch & Prof#=Cottonwood Creek,Reach-1,7
Up Type=0
Dn Type=3
Dn Slope=0.005

--- Cottonwood Creek Trib034.g01 (geometry) ---

Geom Title=Existing Conditions

River Reach=Cottonwood Creek,Reach-1
Reach XY= 30
      1304605.00      6861288.00      1303712.98      6862634.65
      1303405.33      6864372.97      1303597.98      6864778.97
      1304497.49      6864934.82      1304262.08      6865188.00
      1304503.80      6865548.51      1304406.63      6866081.96
      1304905.47      6866467.85      1304113.02      6868591.31
      1304506.17      6869134.88      1304801.31      6868845.65
      1305091.61      6869024.67      1305049.17      6869490.84
      1304756.73      6869631.84      1305370.09      6870037.81
      1308334.97      6870037.93      1311039.82      6869587.57
      1312102.99      6869935.05      1312884.61      6868707.05
      1313391.47      6868701.38      1313344.62      6868298.80
      1314065.00      6868177.05      1314441.32      6867601.50
      1315511.19      6867180.19      1316752.55      6866093.47
      1318461.06      6865480.52      1319828.47      6864414.99
      1321048.81      6862995.85      1321855.00      6862988.00

Type RM Length L Ch R = 1,36179,226,226,226
BEGIN DESCRIPTION:
Cottonwood Creek Trib034 71.0
END DESCRIPTION:
XS GIS Cut Line= 6
      1303666.24      6859175.94      1303785.60      6861200.68
      1304434.47      6861289.66      1304586.38      6861333.06
      1305370.52      6861535.61      1306745.43      6860557.33
#Sta/Elev= 30
  2221.0 2401.62  2683.9 2400.43  2693.9 2397.82  2703.9 2397.67  3515.3 2395.52
  3565.4 2394.39  3845.9 2393.84  4170.3 2391.30  4522.0 2389.34  4773.5 2388.20
  4803.8 2386.72  4874.5 2386.14  5203.4 2385.26  5203.6 2384.76  5207.4 2385.26
  5401.9 2385.85  5708.0 2388.22  6067.2 2390.89  6188.8 2392.40  6209.7 2393.83
  6218.3 2391.29  6239.2 2391.79  6245.8 2393.49  6282.6 2392.67  6295.8 2394.65
  6369.7 2394.11  7192.2 2399.44  7221.7 2400.70  7264.4 2399.93  7559.5 2402.13
#Mann=9,-1,0
  2221.0   0.045       0  4170.3    0.07       0  4522.0   0.045       0
  5203.4   0.045       0  5207.4   0.045       0  5401.9    0.07       0
  5708.0   0.045       0  6067.2   0.035       0  6369.7   0.045       0
Bank Sta=5203.4,5207.4
Exp/Cntr=0.3,0.1

Type RM Length L Ch R = 1,35953,330,330,330
BEGIN DESCRIPTION:
Cottonwood Creek Trib034 70.0
END DESCRIPTION:
XS GIS Cut Line= 6
      1303624.76      6859051.63      1303644.54      6861276.64
      1304296.67      6861458.29      1304443.26      6861507.15
      1305515.20      6861632.54      1306591.72      6861312.18
#Sta/Elev= 30
  1984.6 2401.83  2574.9 2400.11  2961.0 2396.45  3471.0 2395.71  4148.3 2391.48
  4267.9 2390.60  4543.4 2389.30  4673.5 2388.29  5060.2 2383.80  5156.8 2385.05
  5224.2 2385.38  5244.3 2382.93  5264.6 2382.76  5264.8 2382.26  5268.6 2382.76
  5304.7 2384.78  5349.9 2383.81  5475.9 2384.76  5586.6 2387.23  5750.2 2388.36
  5841.4 2388.82  5957.7 2390.38  6090.0 2392.19  6141.1 2390.44  6188.5 2392.15
  6245.4 2391.86  6276.7 2394.04  6335.2 2393.79  7026.5 2400.57  7243.6 2400.99
#Mann=13,-1,0
  1984.6   0.045       0  4148.3    0.07       0  4267.9   0.035       0
  4543.4    0.07       0  4673.5   0.035       0  5060.2   0.045       0
  5156.8   0.035       0  5264.6   0.035       0  5268.6   0.035       0
  5750.2    0.07       0  5841.4   0.045       0  5957.7   0.035       0
  6335.2   0.045       0
Bank Sta=5264.6,5268.6
Exp/Cntr=0.3,0.1

Type RM Length L Ch R = 1,35623,623,623,623
BEGIN DESCRIPTION:
Cottonwood Creek Trib034 69.5
END DESCRIPTION:
XS GIS Cut Line= 5
      1303581.36      6859299.03      1303609.82      6861354.76
      1304253.26      6861705.68      1304399.86      6861754.55
      1306549.92      6861559.09
#Sta/Elev= 30
  2144.4 2401.16  3103.5 2395.26  3713.5 2394.19  3993.6 2391.50  4053.6 2392.21
  4090.7 2390.81  4135.3 2391.05  4272.7 2389.84  4530.8 2388.32  4604.9 2389.48
  4684.6 2386.14  4832.7 2386.07  4890.6 2383.52  5153.2 2382.70  5263.6 2384.06
  5301.8 2381.63  5302.1 2381.13  5305.8 2381.63  5354.0 2383.78  5414.3 2383.29
  5444.4 2385.31  5548.3 2384.37  5645.2 2386.79  5745.6 2386.04  5815.9 2386.72
  5856.1 2388.92  5874.9 2388.11  6403.5 2393.47  6860.2 2398.81  7246.7 2400.89
#Mann=8,-1,0
  2144.4   0.045       0  4090.7    0.07       0  4135.3   0.035       0
  4272.7   0.045       0  5301.8   0.045       0  5305.8   0.045       0
  5874.9   0.035       0  6403.5   0.045       0
Bank Sta=5301.8,5305.8
Exp/Cntr=0.3,0.1

Type RM Length L Ch R = 1,35000,500,500,500
BEGIN DESCRIPTION:
Cottonwood Creek Trib034 69.0
END DESCRIPTION:
XS GIS Cut Line= 4
      1303455.00      6859187.98      1303492.63      6861409.02
      1304132.43      6862160.62      1306604.97      6861738.01
#Sta/Elev= 30
  1791.6 2401.04  3890.3 2390.91  3988.3 2390.02  4105.8 2390.49  4162.9 2388.63
  4474.8 2387.24  4602.6 2384.17  4659.3 2385.07  4702.1 2382.07  4808.6 2382.50
  4872.3 2380.76  5317.1 2381.91  5342.2 2380.71  5378.0 2382.50  5416.6 2380.20
  5416.8 2379.70  5420.6 2380.20  5469.3 2382.87  5550.4 2382.70  5591.0 2384.72
  5938.3 2386.52  5993.3 2388.59  6118.6 2388.55  6402.6 2391.81  6474.2 2394.04
  6818.2 2395.90  6870.8 2396.53  7234.5 2398.45  7338.4 2400.44  7508.4 2401.20
#Mann=8,-1,0
  1791.6   0.045       0  3890.3   0.035       0  3988.3   0.045       0
  5416.6   0.045       0  5420.6   0.045       0  6818.2    0.07       0
  6870.8   0.035       0  7338.4   0.045       0
Bank Sta=5416.6,5420.6
Exp/Cntr=0.3,0.1

Type RM Length L Ch R = 1,34500,500,500,500
BEGIN DESCRIPTION:
Cottonwood Creek Trib034 68.0
END DESCRIPTION:
XS GIS Cut Line= 4
      1300423.96      6862369.35      1303184.31      6862584.52
      1303916.27      6862526.29      1306204.97      6862138.01
#Sta/Elev= 30
  1497.0 2401.59  1819.0 2401.68  2430.9 2397.91  2601.4 2394.27  2842.1 2392.79
  2872.2 2390.96  2972.5 2391.24  3112.9 2389.94  3163.1 2387.81  3524.2 2385.78
  3915.4 2380.15  4625.6 2378.20  4625.8 2377.70  4629.6 2378.20  5465.3 2380.53
  5485.6 2379.39  5516.0 2381.17  5559.7 2378.75  5627.6 2381.63  5789.9 2382.57
  5850.7 2384.88  5982.6 2385.06  6043.4 2387.50  6152.8 2387.28  6246.3 2389.56
  6530.3 2391.41  6621.6 2393.90  6806.7 2394.70  7118.9 2397.31  7321.4 2398.96
#Mann=5,-1,0
  1497.0   0.045       0  4625.6   0.045       0  4629.6   0.045       0
  6806.7    0.07       0  7118.9   0.045       0
Bank Sta=4625.6,4629.6
Exp/Cntr=0.3,0.1

Type RM Length L Ch R = 1,34000,500,500,500
BEGIN DESCRIPTION:
Cottonwood Creek Trib034 67.0
END DESCRIPTION:
XS GIS Cut Line= 3
      1301255.02      6862888.00      1303754.85      6862851.41
      1306054.95      6862288.01
#Sta/Elev= 30
  2499.9 2399.55  2539.9 2398.09  2809.9 2396.84  2989.9 2393.66  3350.0 2391.11
  3390.0 2389.29  3480.0 2389.50  3551.8 2387.00  3737.8 2384.21  3780.0 2382.39
  4060.1 2379.29  4690.1 2379.12  4780.1 2377.12  4918.1 2376.65  4918.4 2376.15
  4922.1 2376.65  5576.7 2379.29  5607.6 2377.95  5638.5 2380.22  5659.1 2378.07
  5690.0 2377.82  5731.1 2379.90  5823.8 2379.64  5865.0 2381.65  6029.7 2382.83
  6060.6 2384.65  6709.2 2391.40  6774.8 2393.80  7000.9 2395.02  7368.1 2398.22
#Mann=7,-1,0
  2499.9   0.045       0  3551.8    0.07       0  3737.8   0.045       0
  4918.1   0.045       0  4922.1   0.045       0  6774.8    0.07       0
  7000.9   0.045       0
Bank Sta=4918.1,4922.1
Exp/Cntr=0.3,0.1

Type RM Length L Ch R = 1,33500,500,500,500
BEGIN DESCRIPTION:
Cottonwood Creek Trib034 66.0
END DESCRIPTION:
XS GIS Cut Line= 3
      1301654.98      6863388.00      1303675.33      6863268.05
      1305804.98      6862588.01
#Sta/Elev= 30
  2976.1 2395.76  3055.9 2396.39  3326.7 2393.01  3777.5 2383.03  3857.7 2382.91
  3897.7 2381.05  4351.9 2379.20  4575.9 2377.46  4730.9 2375.77  4977.4 2374.97
  4977.7 2374.47  4981.8 2374.97  5188.6 2376.56  5439.6 2376.01  5587.5 2377.95
  5605.8 2376.67  5661.0 2378.07  5713.5 2376.45  5900.7 2378.90  5996.9 2378.60
  6049.4 2381.12  6195.6 2382.18  6259.4 2384.80  6431.4 2386.19  6469.3 2388.67
  6694.1 2389.84  6828.1 2392.85  6898.9 2392.86  7081.1 2394.27  7235.6 2395.80
#Mann=8,-1,0
  2976.1   0.045       0  4351.9   0.035       0  4575.9   0.094       0
  4730.9   0.045       0  4977.4   0.045       0  4981.8   0.045       0
  6898.9    0.07       0  7081.1   0.045       0
Bank Sta=4977.4,4981.8
Exp/Cntr=0.3,0.1

Type RM Length L Ch R = 1,33000,500,500,500
BEGIN DESCRIPTION:
Cottonwood Creek Trib034 65.0
END DESCRIPTION:
XS GIS Cut Line= 3
      1301855.02      6863738.00      1303535.95      6863656.52
      1305554.97      6862788.01
#Sta/Elev= 30
  3317.1 2395.19  3567.4 2390.76  3597.4 2391.47  3647.5 2389.11  3727.6 2388.68
  3787.6 2385.83  3830.3 2385.55  3874.7 2385.18  3947.8 2383.11  3997.9 2383.50
  4047.9 2381.17  4278.2 2380.86  4508.5 2378.41  4618.6 2375.75  4668.7 2376.86
  4718.7 2374.78  4929.0 2375.32  5094.7 2373.87  5095.0 2373.37  5099.2 2373.87
  6194.6 2377.82  6283.5 2379.00  6316.2 2380.81  6475.4 2382.11  6522.4 2385.10
  6575.0 2384.21  6697.2 2386.23  6727.1 2388.57  6795.2 2388.08  7197.9 2394.04
#Mann=5,-1,0
  3317.1   0.045       0  3830.3   0.063       0  3874.7   0.045       0
  5094.7   0.045       0  5099.2   0.045       0
Bank Sta=5094.7,5099.2
Exp/Cntr=0.3,0.1

Type RM Length L Ch R = 1,32500,500,500,500
BEGIN DESCRIPTION:
Cottonwood Creek Trib034 64.0
END DESCRIPTION:
XS GIS Cut Line= 3
      1301658.80      6864277.79      1303455.11      6864071.66
      1305605.04      6862787.98
#Sta/Elev= 30
  3191.9 2393.73  3248.5 2394.64  3317.8 2392.78  3661.2 2391.27  3751.7 2388.85
  3792.0 2389.78  4224.8 2380.77  4325.5 2380.97  4657.7 2377.02  4718.0 2375.05
  4929.4 2375.00  4989.3 2372.96  4989.6 2372.46  4993.8 2372.96  5776.0 2373.85
  5871.4 2376.31  5972.5 2374.94  6432.4 2377.69  6503.8 2378.54  6540.7 2380.63
  6694.5 2381.85  6758.7 2384.81  6921.6 2386.24  6965.0 2388.38  7122.6 2389.22
  7151.3 2389.66  7247.7 2392.34  7432.0 2392.77  7498.0 2394.93  7504.0 2394.67
#Mann=6,-1,0
  3191.9   0.045       0  4989.3   0.045       0  4993.8   0.045       0
  7122.6    0.07       0  7151.3   0.045       0  7498.0    0.07       0
Bank Sta=4989.3,4993.8
Exp/Cntr=0.3,0.1

Type RM Length L Ch R = 1,32000,500,500,500
BEGIN DESCRIPTION:
Cottonwood Creek Trib034 63.0
END DESCRIPTION:
XS GIS Cut Line= 3
      1301629.65      6865267.39      1303542.50      6864475.72
      1305455.02      6863237.98
#Sta/Elev= 30
  2929.8 2397.40  3563.3 2391.47  3616.6 2389.19  3699.1 2389.54  3858.7 2385.28
  3965.1 2385.20  4126.1 2380.76  4225.8 2380.47  4266.8 2378.45  4403.9 2377.78
  4457.1 2375.99  4741.6 2375.69  4794.8 2373.26  5025.6 2371.92  5026.0 2371.42
  5030.5 2371.92  5145.9 2373.25  5780.6 2372.56  5977.1 2373.43  6013.4 2374.99
  6113.0 2374.01  6360.9 2377.89  6490.9 2377.88  6539.6 2380.70  6626.8 2380.11
  6756.7 2384.54  7003.0 2388.01  7098.3 2390.74  7140.6 2389.94  7278.1 2392.06
#Mann=4,-1,0
  2929.8   0.045       0  5025.6   0.045       0  5030.5   0.045       0
  7003.0    0.07       0
Bank Sta=5025.6,5030.5
Exp/Cntr=0.3,0.1

Type RM Length L Ch R = 1,31500,500,500,500
BEGIN DESCRIPTION:
Cottonwood Creek Trib034 62.0
END DESCRIPTION:
XS GIS Cut Line= 3
      1301699.13      6865493.07      1303711.92      6864746.18
      1305605.01      6863637.99
#Sta/Elev= 30
  2853.1 2397.41  3296.7 2393.06  3368.4 2393.57  3459.5 2390.93  3499.3 2391.98
  3552.7 2389.55  3638.0 2389.68  3734.0 2386.68  3904.7 2385.15  4096.7 2379.77
  4176.1 2380.25  4192.6 2378.33  4231.5 2377.54  4610.3 2375.59  4665.8 2372.96
  4736.6 2374.13  4834.9 2371.56  4835.2 2371.06  4839.8 2371.56  6149.7 2373.71
  6257.1 2375.82  6272.8 2377.53  6374.4 2377.02  6433.1 2379.88  6556.3 2380.75
  6637.4 2384.24  6741.7 2384.74  6785.0 2387.16  6986.4 2389.66  7193.6 2392.03
#Mann=4,-1,0
  2853.1   0.045       0  4834.9   0.045       0  4839.8   0.045       0
  6986.4    0.07       0
Bank Sta=4834.9,4839.8
Exp/Cntr=0.3,0.1

Type RM Length L Ch R = 1,31000,500,500,500
BEGIN DESCRIPTION:
Cottonwood Creek Trib034 61.0
END DESCRIPTION:
XS GIS Cut Line= 4
      1301780.33      6865493.07      1304063.27      6864937.52
      1304112.20      6864846.39      1305704.99      6863588.01
#Sta/Elev= 30
  2547.0 2397.43  3117.9 2392.79  3178.1 2390.50  3261.5 2390.50  3457.5 2385.25
  3522.2 2385.53  3622.2 2382.38  3677.8 2382.80  3753.3 2380.11  3902.9 2376.41
  4158.4 2376.11  4278.5 2372.98  4361.9 2373.40  4443.0 2371.46  4443.3 2370.96
  4447.9 2371.46  5847.7 2373.09  5897.4 2375.33  5975.9 2375.68  6004.8 2377.90
  6097.8 2377.29  6161.9 2380.10  6239.8 2380.08  6325.4 2383.46  6381.5 2383.25
  6410.3 2385.30  6460.0 2384.58  6509.7 2387.43  6708.0 2389.76  7029.9 2393.75
#Mann=6,-1,0
  2547.0   0.045       0  3677.8    0.07       0  3753.3   0.045       0
  4443.0   0.045       0  4447.9   0.045       0  6708.0    0.07       0
Bank Sta=4443,4447.9
Exp/Cntr=0.3,0.1

Type RM Length L Ch R = 1,30500,500,500,500
BEGIN DESCRIPTION:
Cottonwood Creek Trib034 60.0
END DESCRIPTION:
XS GIS Cut Line= 3
      1301768.61      6865562.51      1304497.69      6864940.35
      1305955.00      6863988.00
#Sta/Elev= 30
  2200.9 2397.42  2679.3 2394.42  2720.3 2392.45  2822.8 2392.27  2871.3 2389.99
  2956.2 2390.57  3010.6 2387.99  3313.1 2383.26  3443.0 2381.55  3748.8 2375.86
  3933.1 2375.08  4002.9 2372.62  4045.9 2373.84  4094.7 2371.76  4268.4 2371.44
  4268.9 2370.94  4274.0 2371.44  5382.0 2372.34  5614.3 2376.34  5795.3 2377.08
  5822.4 2379.28  5844.9 2378.06  5940.1 2378.86  5961.2 2381.04  6012.2 2380.46
  6069.8 2383.38  6112.0 2382.71  6155.5 2385.37  6427.2 2390.08  6740.9 2393.87
#Mann=8,-1,0
  2200.9   0.045       0  3313.1    0.07       0  3443.0   0.045       0
  3748.8    0.07       0  3933.1   0.045       0  4268.4   0.045       0
  4274.0   0.045       0  6427.2    0.07       0
Bank Sta=4268.4,4274
Exp/Cntr=0.3,0.1

Type RM Length L Ch R = 1,30000,500,500,500
BEGIN DESCRIPTION:
Cottonwood Creek Trib034 59.0
END DESCRIPTION:
XS GIS Cut Line= 3
      1301803.27      6865614.61      1304354.14      6865287.17
      1306255.02      6864187.99
#Sta/Elev= 30
  2428.2 2397.24  2903.8 2394.71  2964.3 2392.23  3045.0 2392.88  3105.4 2390.20
  3317.2 2388.32  3385.8 2385.68  3468.4 2385.85  3673.3 2378.72  3912.0 2377.62
  3972.4 2375.52  4083.3 2375.32  4194.3 2372.34  4615.0 2371.27  4615.4 2370.77
  4620.6 2371.27  5578.6 2372.01  5717.2 2374.82  5821.2 2374.36  5855.8 2376.81
  6156.1 2376.67  6201.8 2379.19  6223.3 2378.05  6384.1 2380.73  6411.4 2383.39
  6470.2 2383.04  6501.8 2385.51  6668.3 2389.14  6891.4 2391.06  7195.8 2393.42
#Mann=8,-1,0
  2428.2   0.045       0  3385.8    0.07       0  3673.3   0.045       0
  3972.4    0.07       0  4083.3   0.045       0  4615.0   0.045       0
  4620.6   0.045       0  6891.4    0.07       0
Bank Sta=4615,4620.6
Exp/Cntr=0.3,0.1

Type RM Length L Ch R = 1,29500,500,500,500
BEGIN DESCRIPTION:
Cottonwood Creek Trib034 58.0
END DESCRIPTION:
XS GIS Cut Line= 3
      1301803.31      6865649.33      1304472.96      6865720.60
      1306055.03      6864337.97
#Sta/Elev= 30
  2329.4 2397.35  2921.3 2392.50  2991.3 2393.37  3229.1 2387.70  3451.5 2385.09
  3501.5 2381.77  3591.8 2381.31  3641.6 2378.42  3741.9 2378.20  3955.6 2374.34
  4131.7 2372.06  4739.0 2370.66  4739.5 2370.16  4744.8 2370.66  5825.8 2372.60
  5853.3 2374.80  5981.5 2374.52  6016.6 2376.99  6335.5 2376.68  6378.2 2379.37
  6406.7 2378.07  6470.3 2378.69  6498.8 2381.17  6533.9 2380.03  6583.3 2383.23
  6647.8 2383.31  6676.1 2385.66  6832.0 2388.96  7073.4 2391.17  7101.1 2391.64
#Mann=8,-1,0
  2329.4   0.045       0  3229.1    0.07       0  3591.8   0.045       0
  3741.9    0.07       0  3955.6   0.045       0  4739.0   0.045       0
  4744.8   0.045       0  7073.4    0.07       0
Bank Sta=4739,4744.8
Exp/Cntr=0.3,0.1

Type RM Length L Ch R = 1,29000,1000,1000,1000
BEGIN DESCRIPTION:
Cottonwood Creek Trib034 57.0
END DESCRIPTION:
XS GIS Cut Line= 3
      1301785.94      6865716.17      1304461.84      6866144.72
      1306355.01      6864287.99
#Sta/Elev= 30
  2290.0 2397.42  2886.6 2394.97  3284.2 2388.66  3299.8 2387.06  3470.2 2381.96
  3526.0 2382.03  3585.4 2378.92  3844.3 2376.13  3938.1 2374.65  4487.5 2370.68
  5562.6 2370.48  5563.1 2369.98  5568.5 2370.48  6103.0 2372.57  6138.5 2375.13
  6265.6 2374.51  6301.1 2377.14  6322.2 2375.76  6633.4 2376.94  6661.7 2379.44
  6753.7 2378.65  6796.1 2381.13  6845.5 2380.88  6888.0 2383.38  6944.5 2383.14
  6979.8 2385.72  7029.4 2385.29  7142.6 2388.88  7502.8 2392.14  7651.7 2393.84
#Mann=8,-1,0
  2290.0   0.045       0  3299.8    0.07       0  3526.0   0.045       0
  3844.3    0.07       0  3938.1   0.045       0  5562.6   0.045       0
  5568.5   0.045       0  7502.8    0.07       0
Bank Sta=5562.6,5568.5
Exp/Cntr=0.3,0.1

Type RM Length L Ch R = 1,28000,500,500,500
BEGIN DESCRIPTION:
Cottonwood Creek Trib034 56.0
END DESCRIPTION:
XS GIS Cut Line= 4
      1301759.88      6865872.42      1304789.74      6866502.60
      1304908.63      6866516.69      1306470.28      6864543.40
#Sta/Elev= 30
  1905.3 2397.46  2462.1 2395.71  2778.7 2392.16  2847.4 2389.41  2893.2 2389.75
  2921.7 2386.74  3123.6 2381.68  3188.7 2378.64  3465.3 2376.57  3580.7 2374.39
  3984.0 2370.98  5191.5 2369.49  5192.0 2368.99  5197.6 2369.49  5208.1 2371.09
  5971.0 2370.97  6012.7 2373.17  6134.5 2372.69  6163.4 2374.99  6298.0 2374.58
  6326.8 2377.06  6597.4 2376.65  6639.3 2379.45  6775.6 2379.09  6802.8 2381.16
  6875.0 2380.96  6988.7 2383.41  7024.0 2386.01  7201.9 2388.91  7636.2 2392.18
#Mann=7,-1,0
  1905.3   0.045       0  2847.4    0.07       0  3123.6   0.045       0
  3465.3    0.07       0  3580.7   0.045       0  5191.5   0.045       0
  5197.6   0.045       0
Bank Sta=5191.5,5197.6
Exp/Cntr=0.3,0.1

Type RM Length L Ch R = 1,27500,500,500,500
BEGIN DESCRIPTION:
Cottonwood Creek Trib034 55.0
END DESCRIPTION:
XS GIS Cut Line= 4
      1301629.63      6866028.65      1304654.27      6866925.13
      1306076.96      6866194.86      1307548.33      6862627.12
#Sta/Elev= 30
  1845.3 2397.79  2636.0 2394.13  2925.2 2389.32  3082.4 2382.45  4256.5 2369.90
  4257.0 2369.40  4264.0 2369.90  4320.7 2370.39  4326.0 2373.85  4359.2 2370.37
  4865.4 2370.06  4913.7 2370.10  5080.8 2370.38  5142.7 2370.39  5226.2 2370.53
  5542.8 2370.33  6475.4 2372.60  6492.0 2373.73  6507.0 2380.39  6552.0 2373.64
  6662.8 2373.78  7612.6 2389.06  8425.4 2392.87  8537.9 2393.61  8646.8 2394.15
  8759.1 2394.43  8977.4 2395.06  9467.1 2397.46  9637.0 2398.15 10458.4 2401.94
#Mann=18,-1,0
  1845.3   0.045       0  2636.0    0.07       0  3082.4   0.045       0
  4256.5   0.045       0  4264.0   0.045       0  4865.4    0.07       0
  4913.7   0.045       0  5080.8    0.07       0  5142.7   0.045       0
  5226.2    0.07       0  5542.8   0.045       0  8425.4    0.07       0
  8537.9   0.045       0  8646.8    0.07       0  8759.1   0.045       0
  8977.4    0.07       0  9467.1   0.045       0  9637.0    0.07       0
Bank Sta=4256.5,4264
Exp/Cntr=0.3,0.1

Type RM Length L Ch R = 1,27000,500,500,500
BEGIN DESCRIPTION:
Cottonwood Creek Trib034 54.0
END DESCRIPTION:
XS GIS Cut Line= 4
      1301551.52      6866289.07      1304513.62      6867332.18
      1306310.50      6866427.40      1307626.44      6862835.48
#Sta/Elev= 30
  1859.6 2397.19  2584.2 2394.62  2720.0 2392.37  2912.9 2390.22  3093.4 2384.47
  3225.9 2379.75  3648.7 2374.65  3674.4 2372.77  4640.7 2370.04  4744.0 2370.14
  4820.4 2369.85  4820.9 2369.35  4827.9 2369.85  5695.8 2370.54  5701.9 2370.54
  5944.2 2370.70  6001.8 2370.58  6709.6 2372.28  6770.5 2374.95  6955.1 2374.76
  6983.3 2376.98  7388.8 2378.75  7566.5 2383.52  8033.6 2389.12  9082.5 2393.38
  9289.2 2394.12  9657.6 2395.39  9886.1 2396.52 10279.0 2398.36 10837.2 2401.09
#Mann=16,-1,0
  1859.6   0.045       0  2720.0    0.07       0  3093.4   0.045       0
  4640.7    0.07       0  4744.0   0.045       0  4820.4   0.045       0
  4827.9   0.045       0  5695.8   0.035       0  5701.9   0.045       0
  5944.2    0.07       0  6001.8   0.045       0  9082.5    0.07       0
  9289.2   0.045       0  9657.6    0.07       0  9886.1   0.045       0
 10279.0    0.07       0
Bank Sta=4820.4,4827.9
Exp/Cntr=0.3,0.1

Type RM Length L Ch R = 1,26500,500,500,500
BEGIN DESCRIPTION:
Cottonwood Creek Trib034 53.0
END DESCRIPTION:
XS GIS Cut Line= 4
      1301421.32      6866601.58      1304409.47      6867730.80
      1306315.42      6866815.35      1307730.32      6863135.71
#Sta/Elev= 30
  1805.6 2398.20  2683.7 2393.69  3164.7 2385.27  3365.2 2377.67  3637.6 2373.89
  4913.6 2369.00  4914.1 2368.50  4922.8 2369.00  5787.0 2370.29  6186.7 2370.97
  6187.0 2370.97  6298.2 2371.14  6400.7 2371.39  6408.7 2371.47  6969.7 2374.35
  7023.5 2376.94  7515.3 2376.92  7545.3 2379.47  7878.5 2381.72  7903.2 2384.95
  7933.2 2382.20  8429.4 2388.99  9796.1 2394.06  9870.2 2394.45  9921.2 2394.71
 10298.4 2395.84 10400.4 2396.41 10596.8 2397.43 10608.0 2397.69 11056.7 2399.70
#Mann=16,-1,0
  1805.6   0.045       0  4913.6   0.045       0  4922.8   0.045       0
  5787.0   0.035       0  6186.7   0.045       0  6187.0    0.07       0
  6298.2   0.045       0  6400.7    0.07       0  6408.7   0.045       0
  9796.1    0.07       0  9870.2   0.045       0  9921.2    0.07       0
 10298.4   0.045       0 10400.4    0.07       0 10596.8   0.045       0
 10608.0    0.07       0
Bank Sta=4913.6,4922.8
Exp/Cntr=0.3,0.1

Type RM Length L Ch R = 1,26000,500,500,500
BEGIN DESCRIPTION:
Cottonwood Creek Trib034 52.0
END DESCRIPTION:
XS GIS Cut Line= 4
      1301108.82      6867122.41      1304255.26      6868117.01
      1306493.63      6867054.23      1308081.81      6863292.07
#Sta/Elev= 30
  1700.1 2401.27  2859.1 2393.40  3026.0 2390.51  3090.6 2386.86  3160.5 2386.74
  3198.1 2383.73  3237.8 2384.20  3269.3 2381.33  3405.6 2378.07  3788.3 2374.86
  3859.6 2373.60  4450.4 2370.20  4490.1 2370.09  4764.5 2369.47  5017.1 2368.19
  5017.6 2367.69  5026.6 2368.19  6365.7 2371.11  6626.1 2374.49  6677.9 2374.09
  7039.2 2376.61  7312.7 2376.83  7391.9 2379.42  7827.5 2379.09  8522.0 2387.60
  9700.4 2391.28  9783.1 2391.52 10335.4 2393.80 11048.0 2396.65 11561.5 2399.64
#Mann=16,-1,0
  1700.1   0.045       0  3788.3    0.07       0  3859.6   0.045       0
  4450.4   0.035       0  4490.1   0.063       0  4764.5   0.045       0
  5017.1   0.045       0  5026.6   0.045       0  6365.7    0.07       0
  6626.1   0.045       0  6677.9    0.07       0  7039.2   0.045       0
  9700.4   0.035       0  9783.1   0.045       0 10335.4   0.035       0
 11048.0   0.045       0
Bank Sta=5017.1,5026.6
Exp/Cntr=0.3,0.1

Type RM Length L Ch R = 1,25500,500,500,500
BEGIN DESCRIPTION:
Cottonwood Creek Trib034 51.0
END DESCRIPTION:
XS GIS Cut Line= 4
      1300822.42      6867434.93      1304139.07      6868552.87
      1306594.08      6867201.35      1308537.92      6862926.59
#Sta/Elev= 30
  1500.0 2401.91  2214.5 2399.64  2769.1 2395.31  3159.5 2386.10  3337.4 2379.59
  3724.2 2376.15  4290.8 2370.59  4322.6 2370.63  4900.7 2367.95  5386.7 2367.68
  5387.2 2367.18  5396.2 2367.68  5634.2 2368.94  5899.1 2369.70  6288.3 2370.37
  6578.5 2372.61  6760.6 2376.07  6969.1 2376.89  7107.3 2378.38  7657.3 2379.50
  7733.1 2381.48  7800.7 2379.94  7842.7 2381.22  8130.5 2380.93  8256.8 2383.26
  8763.1 2387.29  9952.3 2390.44 10536.9 2392.60 11634.1 2397.01 12498.4 2404.80
#Mann=14,-1,0
  1500.0   0.045       0  3724.2    0.07       0  4290.8   0.035       0
  4322.6   0.045       0  5386.7   0.045       0  5396.2   0.045       0
  5634.2   0.094       0  5899.1   0.045       0  6288.3    0.07       0
  6578.5   0.045       0  6969.1    0.07       0  7107.3   0.045       0
  9952.3   0.035       0 10536.9   0.045       0
Bank Sta=5386.7,5396.2
Exp/Cntr=0.3,0.1

Type RM Length L Ch R = 1,25000,1500,1500,1500
BEGIN DESCRIPTION:
Cottonwood Creek Trib034 50.0
END DESCRIPTION:
XS GIS Cut Line= 4
      1300614.02      6867695.32      1304387.28      6868920.24
      1306780.09      6867275.59      1308733.08      6862822.77
#Sta/Elev= 30
  1032.9 2402.34  2225.5 2398.55  2550.4 2394.96  2694.3 2390.24  2778.8 2387.89
  2989.5 2380.41  3297.7 2376.58  3895.2 2371.54  4765.5 2367.00  4877.8 2366.71
  4961.3 2366.49  4961.8 2365.99  4970.8 2366.49  5432.8 2369.07  5541.6 2369.70
  5789.5 2371.14  5938.0 2372.00  6260.9 2373.88  6567.5 2375.66  6658.5 2378.63
  6781.1 2381.25  6933.5 2382.53  7222.3 2381.27  8225.0 2384.23  8602.8 2387.32
  9214.7 2388.27  9990.9 2389.96 10903.8 2392.59 11897.4 2398.01 12765.8 2406.83
#Mann=20,-1,0
  1032.9   0.045       0  2694.3    0.07       0  2778.8   0.045       0
  3297.7    0.07       0  3895.2   0.045       0  4765.5   0.035       0
  4877.8    0.07       0  4961.3    0.07       0  4970.8    0.07       0
  5432.8   0.035       0  5541.6   0.045       0  5789.5   0.094       0
  5938.0   0.045       0  6260.9    0.07       0  6658.5   0.035       0
  6781.1    0.07       0  6933.5    0.07       0  7222.3   0.045       0
  9214.7   0.035       0  9990.9   0.045       0
Bank Sta=4961.3,4970.8
Exp/Cntr=0.3,0.1

Type RM Length L Ch R = 1,23500,1000,1000,1000
BEGIN DESCRIPTION:
Cottonwood Creek Trib034 47.0
END DESCRIPTION:
XS GIS Cut Line= 5
      1299200.63      6870950.34      1304233.84      6869440.13
      1305104.64      6869352.44      1306884.25      6867366.73
      1309019.68      6862874.53
#Sta/Elev= 30
 -1130.1 2400.30   183.8 2395.47   705.8 2388.91   980.7 2381.77  1260.8 2377.95
  1964.4 2374.76  2398.8 2371.60  2836.6 2368.59  3230.2 2366.90  3690.1 2366.06
  3690.6 2365.56  3699.9 2366.06  4325.0 2366.39  4405.1 2366.39  4592.7 2366.38
  4879.9 2366.37  4968.0 2366.36  5374.2 2368.32  5776.4 2370.45  6143.7 2372.89
  6738.1 2386.65  7742.6 2386.33  7786.9 2384.37  8286.8 2387.07  8954.4 2388.10
  9178.3 2388.45  9341.8 2388.70 10859.0 2393.84 11943.5 2399.29 12640.4 2406.81
#Mann=20,-1,0
 -1130.1   0.045       0  1964.4    0.07       0  2398.8   0.045       0
  2836.6   0.035       0  3230.2   0.035       0  3690.1   0.045       0
  3699.9   0.035       0  4325.0    0.07       0  4405.1   0.045       0
  4592.7   0.045       0  4879.9   0.035       0  4968.0   0.045       0
  5374.2   0.045       0  5776.4    0.07       0  6738.1   0.045       0
  8286.8   0.035       0  8954.4   0.045       0  9178.3    0.07       0
  9341.8   0.045       0 10859.0   0.045       0
Bank Sta=3690.1,3699.9
Exp/Cntr=0.3,0.1

Type RM Length L Ch R = 1,22500,500,500,500
BEGIN DESCRIPTION:
Cottonwood Creek Trib034 45.0
END DESCRIPTION:
XS GIS Cut Line= 4
      1306267.27      6875615.42      1305071.99      6869704.56
      1306379.21      6868494.34      1309097.02      6862924.58
#Sta/Elev= 30
 -1030.5 2392.87  -736.6 2392.70  -510.7 2392.50  -341.2 2393.57  -285.4 2390.94
   -46.5 2390.21  1779.4 2388.60  1936.7 2387.80  2274.8 2380.33  3155.7 2373.84
  3473.8 2372.52  4158.7 2369.69  5012.9 2365.94  5013.4 2365.44  5028.7 2365.94
  5346.3 2367.42  5622.6 2368.71  6117.8 2371.02  6515.4 2376.12  6781.4 2380.65
  6816.0 2382.59  7055.5 2386.50  7300.3 2388.06  8123.4 2385.35  8491.8 2386.91
  9119.7 2388.22  9954.5 2390.00 11251.6 2393.77 11884.6 2396.51 12978.9 2406.62
#Mann=20,-1,0
 -1030.5    0.07       0  -736.6   0.035       0  -510.7   0.063       0
   -46.5   0.045       0  2274.8    0.07       0  3155.7   0.045       0
  3473.8   0.035       0  4158.7    0.07       0  5012.9   0.035       0
  5028.7   0.035       0  5346.3   0.045       0  5622.6   0.045       0
  6117.8    0.07       0  6515.4   0.045       0  6816.0    0.07       0
  7055.5   0.045       0  8491.8   0.035       0  9119.7   0.045       0
  9954.5   0.045       0 11251.6   0.045       0
Bank Sta=5012.9,5028.7
Exp/Cntr=0.3,0.1

Type RM Length L Ch R = 1,22000,500,500,500
BEGIN DESCRIPTION:
Cottonwood Creek Trib034 44.0
END DESCRIPTION:
XS GIS Cut Line= 4
      1307119.47      6873842.96      1305391.37      6870038.77
      1306419.33      6868549.83      1309072.44      6863047.49
#Sta/Elev= 30
   821.7 2391.02   890.3 2386.83  1000.2 2388.36  2094.5 2389.42  2211.1 2390.31
  2333.3 2388.52  2800.9 2379.56  3760.2 2370.95  4038.9 2367.74  4514.7 2366.18
  4696.1 2366.01  4696.6 2365.51  4712.4 2366.01  5079.2 2366.03  5693.8 2367.06
  6099.6 2370.52  6488.4 2376.03  6793.1 2379.81  6863.5 2382.47  7102.1 2386.42
  7377.5 2387.99  8232.4 2385.36  8404.2 2387.08  9008.0 2387.93  9747.4 2388.69
  9979.5 2388.95 11334.8 2392.87 12373.3 2398.92 12725.6 2404.02 12917.9 2404.57
#Mann=20,-1,0
   821.7   0.063       0  1000.2   0.045       0  2094.5   0.035       0
  2333.3    0.07       0  3760.2   0.035       0  4038.9   0.035       0
  4514.7    0.07       0  4696.1    0.07       0  4712.4    0.07       0
  5079.2   0.035       0  5693.8   0.045       0  6099.6    0.07       0
  6488.4   0.045       0  6863.5    0.07       0  7102.1   0.045       0
  8404.2   0.035       0  9008.0   0.045       0  9747.4   0.045       0
  9979.5   0.045       0 11334.8   0.045       0
Bank Sta=4696.1,4712.4
Exp/Cntr=0.3,0.1

Type RM Length L Ch R = 1,21500,500,500,500
BEGIN DESCRIPTION:
Cottonwood Creek Trib034 43.0
END DESCRIPTION:
XS GIS Cut Line= 3
      1307355.18      6873505.40      1305859.17      6869937.98
      1309019.69      6863226.07
#Sta/Elev= 30
  1131.6 2390.76  1198.0 2387.42  1285.3 2388.95  1918.8 2389.35  2124.4 2389.16
  2394.8 2388.59  2518.8 2389.34  2549.3 2387.29  2859.8 2382.89  3026.4 2378.93
  3518.4 2373.84  3949.5 2370.62  4099.1 2369.35  4987.9 2366.77  4988.4 2366.27
  5004.5 2366.77  5317.7 2368.15  5620.4 2370.36  6114.0 2376.66  6387.0 2378.86
  6529.8 2382.47  6734.3 2385.94  6785.5 2387.85  7122.2 2388.12  7885.2 2386.83
  8460.3 2387.42  9620.4 2388.83 11044.1 2393.28 12022.4 2398.74 12418.8 2403.58
#Mann=20,-1,0
  1131.6   0.063       0  1285.3   0.045       0  1918.8   0.035       0
  2124.4   0.045       0  2394.8    0.07       0  2859.8    0.07       0
  3518.4   0.035       0  3949.5   0.035       0  4099.1   0.045       0
  4987.9   0.045       0  5004.5   0.045       0  5317.7   0.045       0
  5620.4    0.07       0  6114.0   0.045       0  6529.8    0.07       0
  6734.3   0.045       0  7885.2   0.035       0  8460.3   0.045       0
  9620.4   0.045       0 11044.1   0.045       0
Bank Sta=4987.9,5004.5
Exp/Cntr=0.3,0.1

Type RM Length L Ch R = 1,21000,1000,1000,1000
BEGIN DESCRIPTION:
Cottonwood Creek Trib034 42.0
END DESCRIPTION:
XS GIS Cut Line= 3
      1307482.56      6873307.86      1306358.10      6869944.24
      1309152.66      6863022.49
#Sta/Elev= 30
  1453.4 2390.27  1518.0 2387.95  1598.4 2389.13  1950.3 2389.11  2152.1 2389.28
  2567.3 2389.17  2812.9 2388.85  2894.2 2386.80  2964.0 2385.76  3529.8 2377.00
  3708.2 2375.55  3757.7 2374.11  3812.4 2373.83  3916.6 2372.29  4958.7 2370.29
  5071.4 2370.97  5095.4 2369.39  5095.9 2368.89  5112.1 2369.39  5157.7 2372.31
  5692.7 2376.50  5801.5 2376.31  6071.3 2378.97  6500.6 2387.96  7715.3 2387.22
  7821.3 2387.34  9611.6 2388.52 10748.7 2392.40 11908.7 2399.04 12464.6 2405.11
#Mann=20,-1,0
  1453.4   0.063       0  1518.0   0.035       0  1598.4   0.045       0
  1950.3   0.035       0  2152.1   0.045       0  2567.3    0.07       0
  2894.2   0.035       0  2964.0    0.07       0  3529.8   0.035       0
  3708.2    0.07       0  3757.7   0.035       0  3812.4    0.07       0
  3916.6   0.045       0  4958.7    0.07       0  5095.4    0.07       0
  5112.1    0.07       0  5692.7    0.07       0  5801.5   0.045       0
  7715.3   0.035       0  7821.3   0.045       0
Bank Sta=5095.4,5112.1
Exp/Cntr=0.3,0.1

Type RM Length L Ch R = 1,20000,1507,1507,1507
BEGIN DESCRIPTION:
Cottonwood Creek Trib034 40.0
END DESCRIPTION:
XS GIS Cut Line= 3
      1307879.63      6872817.07      1307326.89      6870038.01
      1309152.84      6863104.51
#Sta/Elev= 30
  2166.5 2391.05  2185.9 2389.10  2257.3 2390.64  2318.2 2388.30  2418.6 2389.19
  3582.8 2388.95  3679.5 2387.09  3910.8 2385.82  3980.4 2383.22  4051.8 2383.43
  4115.3 2380.68  4255.7 2379.06  4899.6 2376.29  4907.9 2376.28  4969.4 2377.23
  5000.3 2375.10  5000.8 2374.60  5017.1 2375.10  5044.1 2376.49  5482.1 2378.49
  5650.6 2382.53  5827.4 2384.90  6023.8 2387.76  7559.1 2388.76  7629.3 2388.74
  8664.9 2388.10  9591.4 2390.52  9647.0 2388.85 11349.4 2396.60 12169.9 2404.79
#Mann=13,-1,0
  2166.5   0.063       0  2318.2   0.035       0  2418.6   0.045       0
  3679.5    0.07       0  4899.6   0.045       0  4907.9    0.07       0
  5000.3    0.07       0  5017.1    0.07       0  5044.1   0.045       0
  5650.6    0.07       0  5827.4   0.045       0  7559.1   0.035       0
  7629.3   0.045       0
Bank Sta=5000.3,5017.1
Exp/Cntr=0.3,0.1

Type RM Length L Ch R = 1,18493,791,791,791
BEGIN DESCRIPTION:
Cottonwood Creek Trib034 35.5
END DESCRIPTION:
XS GIS Cut Line= 3
      1308008.80      6872601.86      1308816.15      6870012.02
      1309243.48      6863172.12
#Sta/Elev= 30
  2263.2 2388.64  2297.1 2389.61  2302.4 2388.59  2329.6 2390.42  2334.9 2389.54
  2392.9 2390.91  2502.7 2389.86  2535.2 2388.36  2827.5 2388.88  4613.6 2388.48
  4896.4 2389.68  4916.9 2388.72  4975.5 2388.55  7220.2 2388.51  7334.6 2388.21
  7907.3 2387.98  7907.8 2387.48  7924.1 2387.98  9589.0 2389.68  9969.7 2392.68
  9989.7 2391.90 10270.3 2392.81 11021.8 2396.62 11041.8 2397.61 11129.4 2397.02
 11582.8 2400.48 11610.5 2401.72 11753.2 2402.83 11775.8 2403.86 11829.2 2403.35
#Mann=6,-1,0
  2263.2   0.063       0  2827.5   0.045       0  7220.2   0.035       0
  7334.6   0.045       0  7907.3   0.045       0  7924.1   0.045       0
Bank Sta=7907.3,7924.1
Exp/Cntr=0.3,0.1

Type RM Length L Ch R = 1,17702,702,702,702
BEGIN DESCRIPTION:
Cottonwood Creek Trib034 35.0
END DESCRIPTION:
XS GIS Cut Line= 3
      1308035.90      6872566.99      1309571.31      6869872.65
      1309390.04      6863053.18
#Sta/Elev= 30
  1897.6 2389.49  2087.0 2389.83  2108.6 2388.44  2226.8 2390.58  2775.3 2390.28
  2868.5 2389.41  3149.0 2387.72  3149.5 2387.22  3165.8 2387.72  3329.9 2388.63
  3551.8 2389.10  3796.3 2389.43  4233.6 2390.52  4308.6 2389.14  4367.6 2390.35
  4764.7 2389.15  4883.0 2389.03  4975.4 2388.94  5092.5 2388.60  5767.9 2388.69
  6529.0 2388.37  6979.7 2388.31  7099.1 2388.29  7861.7 2388.21  8241.4 2388.70
  8672.6 2389.57  8908.5 2390.05 10375.3 2393.81 11315.6 2399.31 11820.6 2404.61
#Mann=20,-1,0
  1897.6   0.063       0  2775.3   0.035       0  2868.5   0.063       0
  3149.0   0.035       0  3165.8   0.063       0  3329.9   0.035       0
  3551.8   0.035       0  3796.3   0.035       0  4764.7   0.035       0
  4883.0   0.045       0  4975.4   0.035       0  5092.5   0.045       0
  5767.9   0.035       0  6529.0   0.045       0  6979.7   0.035       0
  7099.1   0.045       0  7861.7    0.07       0  8241.4   0.045       0
  8672.6    0.07       0  8908.5   0.045       0
Bank Sta=3149,3165.8
Exp/Cntr=0.3,0.1

Type RM Length L Ch R = 1,17000,1000,1000,1000
BEGIN DESCRIPTION:
Cottonwood Creek Trib034 34.0
END DESCRIPTION:
XS GIS Cut Line= 3
      1308556.72      6871837.85      1310230.06      6869737.79
      1309963.05      6865901.67
#Sta/Elev= 30
  2314.8 2391.60  2704.9 2390.89  2804.2 2388.41  3555.2 2389.01  3578.3 2389.08
  3700.7 2388.92  3726.4 2389.13  3891.2 2388.86  3978.4 2389.02  4283.2 2389.16
  4552.6 2386.20  4880.5 2376.16  4988.6 2372.53  5136.8 2372.00  5241.9 2370.68
  5242.4 2370.18  5258.8 2370.68  5348.6 2375.56  5434.4 2373.02  5470.9 2375.37
  5606.4 2372.94  5671.4 2378.66  5860.9 2377.55  6251.3 2384.31  6693.9 2388.78
  7577.6 2388.39  7727.1 2388.64  8129.7 2389.22  8749.1 2390.18  8845.4 2390.40
#Mann=20,-1,0
  2314.8   0.035       0  3555.2   0.045       0  3578.3   0.035       0
  3700.7   0.094       0  3726.4   0.035       0  3891.2   0.045       0
  3978.4   0.035       0  4283.2   0.045       0  4552.6   0.035       0
  4880.5   0.045       0  5136.8   0.035       0  5241.9   0.045       0
  5258.8   0.035       0  5348.6   0.063       0  5606.4   0.035       0
  6251.3   0.045       0  7577.6   0.035       0  7727.1    0.07       0
  8129.7   0.035       0  8749.1    0.07       0
Bank Sta=5241.9,5258.8
Exp/Cntr=0.3,0.1

Type RM Length L Ch R = 1,16000,500,500,500
BEGIN DESCRIPTION:
Cottonwood Creek Trib034 32.0
END DESCRIPTION:
XS GIS Cut Line= 3
      1308521.96      6871889.97      1311181.64      6869587.87
      1310015.05      6865848.31
#Sta/Elev= 30
  1482.4 2391.59  1748.6 2387.56  2294.7 2388.83  2547.2 2388.62  3449.7 2388.75
  3613.1 2387.14  3757.2 2381.97  3913.4 2378.08  4215.7 2366.30  4630.7 2360.24
  4940.7 2358.63  5061.8 2358.22  5062.3 2357.72  5078.8 2358.22  5626.0 2361.17
  6060.3 2367.20  6131.2 2370.26  6194.1 2376.46  6314.8 2379.08  6372.1 2376.73
  6406.0 2380.01  6634.0 2386.78  6754.2 2387.64  7434.3 2388.28  7544.2 2388.66
  7647.6 2388.52  7826.5 2388.50  8233.7 2389.16  8585.8 2390.20  8917.3 2390.46
#Mann=20,-1,0
  1482.4   0.035       0  2294.7    0.07       0  2547.2   0.045       0
  3757.2    0.07       0  3913.4   0.045       0  4215.7   0.035       0
  4630.7    0.07       0  4940.7    0.07       0  5061.8    0.07       0
  5078.8    0.07       0  5626.0   0.035       0  6060.3   0.063       0
  6406.0   0.035       0  6754.2   0.045       0  7434.3   0.035       0
  7544.2    0.07       0  7647.6   0.045       0  7826.5    0.07       0
  8233.7   0.045       0  8585.8   0.035       0
Bank Sta=5061.8,5078.8
Exp/Cntr=0.3,0.1

Type RM Length L Ch R = 1,15500,500,500,500
BEGIN DESCRIPTION:
Cottonwood Creek Trib034 31.0
END DESCRIPTION:
XS GIS Cut Line= 3
      1311920.34      6871828.67      1311596.58      6869727.47
      1310175.56      6865873.82
#Sta/Elev= 30
  2874.0 2386.65  3198.5 2382.18  3267.2 2378.31  3421.1 2376.13  3633.8 2369.10
  3805.5 2367.41  3924.4 2362.09  4182.9 2360.31  4362.7 2358.82  4375.2 2358.77
  4848.5 2357.15  4849.0 2356.65  4867.2 2357.15  5766.0 2358.11  6126.8 2361.55
  6373.3 2365.44  6555.9 2373.39  6587.5 2372.51  6617.4 2376.03  6697.4 2377.46
  6727.9 2381.81  6778.1 2383.32  6808.5 2380.86  6897.1 2385.60  6993.3 2387.00
  7560.4 2388.55  7695.2 2388.51  7865.8 2388.53  7920.2 2388.78  9107.3 2390.85
#Mann=15,-1,0
  2874.0   0.045       0  3633.8   0.035       0  4182.9    0.07       0
  4362.7   0.035       0  4375.2    0.07       0  4848.5    0.07       0
  4867.2    0.07       0  6126.8   0.035       0  6617.4   0.063       0
  6897.1   0.035       0  6993.3   0.045       0  7560.4   0.035       0
  7695.2   0.045       0  7865.8    0.07       0  7920.2   0.045       0
Bank Sta=4848.5,4867.2
Exp/Cntr=0.3,0.1

Type RM Length L Ch R = 1,15000,558,558,558
BEGIN DESCRIPTION:
Cottonwood Creek Trib034 30.0
END DESCRIPTION:
XS GIS Cut Line= 3
      1312595.25      6872073.88      1311922.35      6869805.69
      1310142.99      6865737.06
#Sta/Elev= 30
  2634.1 2387.90  2744.6 2387.28  2954.3 2386.28  3145.5 2384.02  3605.9 2369.12
  3884.3 2363.62  4100.7 2361.73  4650.1 2357.91  4894.3 2356.97  5047.1 2356.83
  5047.6 2356.33  5066.1 2356.83  5197.9 2357.33  6189.4 2359.01  6576.4 2363.55
  6680.9 2366.90  6722.0 2370.50  6765.6 2370.19  6885.7 2375.06  6915.6 2378.30
  6978.0 2378.13  7016.7 2383.47  7065.9 2384.38  7093.1 2382.24  7123.8 2385.45
  7213.5 2387.15  7697.7 2388.59  7805.5 2388.71  9388.1 2391.27  9440.7 2391.35
#Mann=18,-1,0
  2634.1   0.045       0  2744.6    0.07       0  2954.3   0.045       0
  3605.9   0.035       0  3884.3    0.07       0  4100.7   0.035       0
  4650.1    0.07       0  4894.3   0.045       0  5047.1   0.045       0
  5066.1   0.045       0  5197.9    0.07       0  6189.4   0.035       0
  6915.6   0.063       0  7065.9   0.035       0  7213.5   0.045       0
  7697.7   0.035       0  7805.5   0.045       0  9388.1   0.035       0
Bank Sta=5047.1,5066.1
Exp/Cntr=0.3,0.1

Type RM Length L Ch R = 1,14442,531,531,531
BEGIN DESCRIPTION:
Cottonwood Creek Trib034 29.0
END DESCRIPTION:
XS GIS Cut Line= 3
      1313409.04      6872084.71      1312235.22      6869709.15
      1310186.39      6865737.06
#Sta/Elev= 30
  2348.5 2387.72  2353.6 2387.71  2648.0 2386.60  2835.6 2386.58  2968.3 2383.50
  3081.0 2381.98  3114.2 2379.35  3517.8 2367.78  3722.5 2363.88  4232.3 2359.49
  4625.4 2357.72  4830.8 2357.01  5147.3 2356.74  5147.8 2356.24  5166.5 2356.74
  5605.5 2357.18  6227.4 2358.67  6423.4 2360.28  6707.7 2364.20  6735.5 2367.04
  6832.4 2370.16  7012.3 2376.29  7066.1 2380.41  7114.9 2380.28  7159.9 2385.28
  7217.3 2383.45  7279.0 2387.20  7676.5 2388.63  7802.2 2388.67  9467.6 2390.91
#Mann=20,-1,0
  2348.5   0.045       0  2353.6    0.07       0  2648.0   0.045       0
  2968.3   0.035       0  3114.2   0.045       0  3517.8   0.035       0
  3722.5    0.07       0  4232.3   0.035       0  4625.4    0.07       0
  4830.8   0.045       0  5147.3   0.045       0  5166.5   0.045       0
  5605.5    0.07       0  6227.4   0.035       0  6423.4   0.035       0
  6832.4   0.035       0  7066.1   0.063       0  7279.0   0.045       0
  7676.5   0.035       0  7802.2   0.045       0
Bank Sta=5147.3,5166.5
Exp/Cntr=0.3,0.1

Type RM Length L Ch R = 1,13911,411,411,411
BEGIN DESCRIPTION:
Cottonwood Creek Trib034 28.0
END DESCRIPTION:
XS GIS Cut Line= 3
      1314277.09      6871520.47      1312498.33      6869484.22
      1310284.06      6865747.93
#Sta/Elev= 30
  2210.3 2382.27  2665.4 2380.51  2672.5 2380.10  2780.7 2379.10  3106.2 2369.72
  3390.2 2363.59  3651.7 2361.08  4268.6 2358.97  4376.7 2357.76  4620.1 2357.05
  4854.6 2356.77  4855.1 2356.27  4873.9 2356.77  5493.7 2356.96  6100.4 2358.45
  6256.3 2359.54  6552.2 2364.96  6759.1 2370.16  6876.1 2376.96  6928.8 2377.41
  6988.6 2382.41  7024.3 2381.52  7051.5 2385.42  7088.6 2386.71  7113.5 2385.14
  7189.9 2388.21  7294.5 2388.16  7397.8 2388.58  7590.5 2388.44  9257.2 2390.96
#Mann=20,-1,0
  2210.3   0.045       0  2665.4    0.07       0  2672.5   0.045       0
  3106.2   0.035       0  3390.2    0.07       0  3651.7   0.035       0
  4268.6   0.035       0  4376.7    0.07       0  4620.1   0.045       0
  4854.6   0.045       0  4873.9   0.045       0  5493.7    0.07       0
  6100.4   0.035       0  6256.3    0.07       0  6552.2   0.035       0
  6988.6   0.063       0  7113.5   0.035       0  7294.5   0.045       0
  7397.8   0.035       0  7590.5   0.045       0
Bank Sta=4854.6,4873.9
Exp/Cntr=0.3,0.1

Type RM Length L Ch R = 1,13500,500,500,500
BEGIN DESCRIPTION:
Cottonwood Creek Trib034 27.0
END DESCRIPTION:
XS GIS Cut Line= 3
      1314255.00      6871038.00      1312660.49      6869132.14
      1310404.25      6865781.72
#Sta/Elev= 30
  2515.1 2381.56  2583.5 2378.93  2714.2 2375.60  2975.6 2367.88  3231.2 2363.78
  3747.4 2359.68  3929.5 2358.75  4357.0 2357.45  4544.2 2358.25  4846.9 2357.21
  5185.1 2356.81  5185.6 2356.31  5204.5 2356.81  5261.0 2356.98  5785.5 2358.23
  5938.1 2358.56  6092.2 2360.20  6372.1 2363.74  6499.3 2364.65  6535.3 2367.94
  6584.3 2367.94  6690.3 2373.45  6850.2 2379.35  6895.3 2383.37  6946.0 2382.88
  6967.1 2386.39  7003.1 2387.69  7039.1 2385.48  7106.9 2388.73  9039.3 2390.92
#Mann=20,-1,0
  2515.1    0.07       0  2583.5   0.063       0  2714.2    0.07       0
  2975.6   0.035       0  3231.2    0.07       0  3747.4   0.035       0
  3929.5    0.07       0  4357.0    0.07       0  4544.2   0.094       0
  4846.9   0.045       0  5185.1   0.045       0  5204.5   0.045       0
  5261.0    0.07       0  5785.5   0.035       0  5938.1    0.07       0
  6092.2   0.045       0  6372.1    0.07       0  6690.3   0.035       0
  6895.3   0.063       0  7106.9   0.045       0
Bank Sta=5185.1,5204.5
Exp/Cntr=0.3,0.1

Type RM Length L Ch R = 1,13000,500,500,500
BEGIN DESCRIPTION:
Cottonwood Creek Trib034 26.0
END DESCRIPTION:
XS GIS Cut Line= 3
      1314755.01      6870638.01      1312855.68      6868754.35
      1310436.99      6865781.73
#Sta/Elev= 30
  2325.0 2381.55  2419.0 2378.98  2554.5 2374.24  2607.8 2373.45  2653.4 2369.90
  2843.7 2366.37  3023.2 2363.84  3543.4 2359.63  3705.3 2358.54  4091.6 2357.96
  4327.0 2357.73  4455.9 2357.36  4669.2 2356.87  4776.0 2356.83  4776.5 2356.33
  4795.5 2356.83  5206.5 2357.06  5723.1 2358.64  6070.7 2361.46  6326.9 2366.46
  6560.4 2375.41  6689.6 2380.51  6724.4 2384.14  6774.4 2383.22  6803.0 2387.10
  6838.8 2387.84  6874.9 2385.83  6924.4 2388.91  6962.6 2388.07  8832.3 2391.08
#Mann=20,-1,0
  2325.0    0.07       0  2419.0   0.063       0  2554.5   0.063       0
  2653.4   0.035       0  2843.7   0.035       0  3023.2    0.07       0
  3543.4   0.035       0  3705.3    0.07       0  4091.6   0.035       0
  4327.0    0.07       0  4455.9    0.07       0  4669.2   0.045       0
  4776.0   0.045       0  4795.5   0.045       0  5206.5   0.035       0
  5723.1   0.045       0  6070.7    0.07       0  6560.4   0.035       0
  6724.4   0.063       0  6962.6   0.045       0
Bank Sta=4776,4795.5
Exp/Cntr=0.3,0.1

Type RM Length L Ch R = 1,12500,500,500,500
BEGIN DESCRIPTION:
Cottonwood Creek Trib034 25.0
END DESCRIPTION:
XS GIS Cut Line= 3
      1314855.00      6870588.00      1313248.66      6868836.45
      1310544.44      6865737.03
#Sta/Elev= 30
  2623.4 2381.92  2834.9 2376.33  3083.7 2367.18  3189.8 2367.00  3345.8 2363.11
  3896.6 2359.48  4022.5 2359.18  4396.0 2357.94  4776.6 2357.27  4866.9 2358.50
  4908.0 2356.90  5253.6 2356.81  5254.1 2356.31  5273.2 2356.81  5309.7 2356.93
  5451.8 2357.41  5867.3 2358.37  5989.7 2358.29  6181.7 2359.86  6602.5 2366.43
  6859.7 2375.81  6950.2 2380.22  7007.2 2380.90  7042.8 2384.25  7099.2 2383.50
  7127.7 2387.59  7179.0 2386.51  7240.8 2388.67  7307.5 2387.71  9113.3 2391.13
#Mann=20,-1,0
  2623.4    0.07       0  2834.9   0.035       0  3345.8    0.07       0
  3896.6   0.035       0  4022.5    0.07       0  4396.0   0.035       0
  4776.6    0.07       0  4908.0   0.045       0  5253.6   0.045       0
  5273.2   0.045       0  5309.7   0.035       0  5451.8    0.07       0
  5867.3   0.045       0  5989.7   0.035       0  6181.7   0.045       0
  6602.5    0.07       0  6859.7   0.035       0  7042.8   0.063       0
  7179.0   0.035       0  7307.5   0.045       0
Bank Sta=5253.6,5273.2
Exp/Cntr=0.3,0.1
