--- BULL WAGON CREEK.prj (project) ---

Proj Title=BULL WAGON CREEK Base Level Engineering
Current Plan=p01
Default Exp/Contr=0.3,0.1
English Units
Geom File=g01
Flow File=f01
Plan File=p01
Y Axis Title=Elevation
X Axis Title(PF)=Main Channel Distance
X Axis Title(XS)=Station
BEGIN DESCRIPTION:
BULL WAGON CREEK
END DESCRIPTION:
DSS Export Rating Curves= 0
DSS Export Rating Curve Sorted= 0
DSS Export Volume Flow Curves= 0
DXF OffsetX= 0
DXF OffsetY= 0
DXF ScaleX= 1
DXF ScaleY= 10

--- BULL WAGON CREEK.p01 (plan) ---

Plan Title=Multiple Run
Short Identifier=Multiple
Geom File=g01
Flow File=f01
Subcritical Flow
K Sum by GR= 0
Std Step Tol= 0.01
Critical Tol= 0.01
Num of Std Step Trials= 20
Max Error Tol= 0.3
Flow Tol Ratio= 0.001
Split Flow NTrial= 30
Split Flow Tol= 0.02
Split Flow Ratio= 0.02
Log Output Level= 0
Friction Slope Method= 1
Unsteady Friction Slope Method= 2
Unsteady Bridges Friction Slope Method= 1
Parabolic Critical Depth
Global Vel Dist=  1 , 1 , 1
Global Log Level= 0
CheckData=True
Encroach Param= -1, 0, 0, 0
BEGIN DESCRIPTION:
Multiple Run
END DESCRIPTION:

--- BULL WAGON CREEK.f01 (steady flow) ---

Flow Title=Multiple
Program Version=4.10
Number of Profiles= 7
Profile Names=10-year,25-year,50-year,1pct_min,100-year,1pct_plu,500-year
River Rch & RM=BULL WAGON CREEK,Reach-1         ,103812
     360     524     668     424     847    1690    1380
River Rch & RM=BULL WAGON CREEK,Reach-1         ,100901
     562     837    1081     696    1388    2770    2321
River Rch & RM=BULL WAGON CREEK,Reach-1         ,96245
     896    1355    1769    1148    2291    4571    3897
River Rch & RM=BULL WAGON CREEK,Reach-1         ,92004
     862    1294    1679    1083    2161    4312    3630
River Rch & RM=BULL WAGON CREEK,Reach-1         ,84552
    1152    1746    2280    1479    2950    5887    5010
River Rch & RM=BULL WAGON CREEK,Reach-1         ,82023
    1342    2038    2668    1732    3455    6894    5881
River Rch & RM=BULL WAGON CREEK,Reach-1         ,69953
    1464    2224    2911    1889    3769    7519    6407
River Rch & RM=BULL WAGON CREEK,Reach-1         ,62654
    1483    2251    2944    1909    3808    7598    6463
River Rch & RM=BULL WAGON CREEK,Reach-1         ,57523
    1540    2338    3057    1982    3954    7889    6708
River Rch & RM=BULL WAGON CREEK,Reach-1         ,54253
    1571    2384    3116    2018    4027    8036    6826
River Rch & RM=BULL WAGON CREEK,Reach-1         ,49402
    1903    2906    3815    2482    4952    9880    8458
River Rch & RM=BULL WAGON CREEK,Reach-1         ,46980
    1971    3012    3958    2575    5139   10253    8787
River Rch & RM=BULL WAGON CREEK,Reach-1         ,45129
    1991    3040    3992    2596    5180   10336    8847
River Rch & RM=BULL WAGON CREEK,Reach-1         ,41815
    2024    3088    4052    2633    5254   10483    8959
River Rch & RM=BULL WAGON CREEK,Reach-1         ,36334
    2017    3070    4022    2609    5206   10387    8845
River Rch & RM=BULL WAGON CREEK,Reach-1         ,29116
    2054    3127    4097    2658    5304   10584    9014
River Rch & RM=BULL WAGON CREEK,Reach-1         ,26898
    2072    3152    4127    2676    5339   10652    9059
River Rch & RM=BULL WAGON CREEK,Reach-1         ,22601
    2064    3137    4104    2659    5305   10584    8986
River Rch & RM=BULL WAGON CREEK,Reach-1         ,18712
    2055    3118    4077    2639    5265   10505    8904
River Rch & RM=BULL WAGON CREEK,Reach-1         ,13610
    2102    3192    4175    2703    5394   10762    9128
River Rch & RM=BULL WAGON CREEK,Reach-1         ,12661
    2208    3356    4392    2845    5677   11327    9618
River Rch & RM=BULL WAGON CREEK,Reach-1         ,9317
    2255    3428    4487    2907    5800   11572    9827
River Rch & RM=BULL WAGON CREEK,Reach-1         ,7185
    2254    3424    4480    2901    5787   11547    9794
River Rch & RM=BULL WAGON CREEK,Reach-1         ,1718
    2274    3455    4520    2926    5838   11649    9878
Boundary for River Rch & Prof#=BULL WAGON CREEK,Reach-1         , 1
Up Type= 0
Dn Type= 3
Dn Slope=0.0019
Boundary for River Rch & Prof#=BULL WAGON CREEK,Reach-1         , 2
Up Type= 0
Dn Type= 3
Dn Slope=0.0019
Boundary for River Rch & Prof#=BULL WAGON CREEK,Reach-1         , 3
Up Type= 0
Dn Type= 3
Dn Slope=0.0019
Boundary for River Rch & Prof#=BULL WAGON CREEK,Reach-1         , 4
Up Type= 0
Dn Type= 3
Dn Slope=0.0019
Boundary for River Rch & Prof#=BULL WAGON CREEK,Reach-1         , 5
Up Type= 0
Dn Type= 3
Dn Slope=0.0019
Boundary for River Rch & Prof#=BULL WAGON CREEK,Reach-1         , 6
Up Type= 0
Dn Type= 3
Dn Slope=0.0019
Boundary for River Rch & Prof#=BULL WAGON CREEK,Reach-1         , 7
Up Type= 0
Dn Type= 3
Dn Slope=0.0019
DSS Import GetInterval= 0
DSS Import GetPeak= 0
DSS Import FillOption= 0

--- BULL WAGON CREEK.g01 (geometry) ---

Geom Title=Existing Conditions
Program Version=4.10

River Reach=BULL WAGON CREEK,Reach-1
Reach XY= 30
        1516505.        6823638.       1517852.7      6825432.94
      1519544.05      6825177.98      1520555.36       6827212.8
      1519960.68      6830290.39      1524196.23      6834081.15
      1523956.78      6836281.87      1525549.94       6837135.7
      1525462.77      6840541.41      1526854.24      6841748.69
      1525908.37      6842686.26      1528653.03      6845943.67
      1528010.28      6847040.71        1531455.        6848788.
      1532947.52      6850784.43      1532315.18       6851697.7
      1534096.11      6852231.49       1533056.2       6852927.5
      1534652.06      6853496.56      1533554.49      6854362.96
      1534653.38      6855331.96      1532262.67      6857281.47
      1532460.68      6858740.52      1533544.82      6858678.29
      1535498.92      6862480.53      1538735.79      6862768.06
      1540253.56      6865044.43      1539857.93      6867030.03
      1541628.47      6867261.01        1544105.        6871088.

Type RM Length L Ch R = 1 ,103812  ,779,779,779
BEGIN DESCRIPTION:
BULL WAGON CREEK 94.0
END DESCRIPTION:
XS GIS Cut Line= 3
      1515961.39      6823977.28        1516755.        6823738.
      1516999.62      6823303.65
#Sta/Elev= 30
  4175.4 1958.81  4182.7 1958.74  4208.2 1958.64  4329.7 1957.82  4356.7 1956.98
  4400.9 1956.93  4450.7 1955.77  4751.7 1952.25  4795.4 1952.68  4826.7 1951.44
  4837.2 1951.58  4850.6 1952.82  4868.5 1951.76  4876.4 1949.63  4876.6 1949.13
  4880.1 1949.13  4880.4 1949.63  4883.6  1950.9  4899.9 1953.04  4916.6 1951.96
  4949.6 1951.27  4954.8 1951.75  5027.3  1950.6  5107.6 1954.97    5385 1960.41
    5401  1961.2  5422.6 1961.09  5438.6 1961.92  5481.9 1962.43  5502.8 1962.12
#Mann= 6 ,-1 , 0
  4175.4    .035       0  4182.7     .07       0  4208.2    .035       0
  4751.7     .07       0  4876.4     .07       0  4880.4     .07       0
Bank Sta=4876.4,4880.4
XS Rating Curve= 0 ,0
Exp/Cntr=0.3,0.1

Type RM Length L Ch R = 1 ,103033  ,471,471,471
BEGIN DESCRIPTION:
Mapping XS 5332e6e8
END DESCRIPTION:
XS GIS Cut Line= 4
      1515989.16      6824630.06        1516701.      6824380.05
      1517096.83      6824046.71      1517180.08      6823883.69
#Sta/Elev= 30
  4239.2 1954.16  4353.9 1952.84  4384.8 1952.92  4410.5 1952.17  4472.5 1952.05
  4478.6 1951.56  4637.5 1949.93  4690.5 1948.58  4864.7 1945.99  4895.7 1946.35
  4902.5 1945.97  4966.1 1945.83  5017.3  1944.9  5017.6  1944.4  5021.1  1944.4
  5021.3  1944.9  5033.6 1946.01  5047.9 1945.39  5062.2 1946.76  5103.9 1946.65
  5132.5 1947.35  5140.2 1947.03  5161.1 1947.84  5218.3 1946.44  5232.6 1947.02
  5352.3 1946.24  5444.6 1947.21  5466.7 1946.92  5655.7 1949.19  5694.2 1948.99
#Mann= 4 ,-1 , 0
  4239.2    .035       0  4966.1     .07       0  5017.3     .07       0
  5021.3     .07       0
Bank Sta=5017.3,5021.3
XS Rating Curve= 0 ,0
Exp/Cntr=0.3,0.1

Type RM Length L Ch R = 1 ,102562  ,556,556,556
BEGIN DESCRIPTION:
BULL WAGON CREEK 93.0
END DESCRIPTION:
XS GIS Cut Line= 3
      1516082.98      6824883.51      1516931.62      6824764.82
      1517357.07      6823852.66
#Sta/Elev= 30
  4143.1 1952.28  4277.2 1950.36  4722.6 1945.89  4902.4 1944.42  5014.4  1942.4
  5014.7  1941.9  5018.2  1941.9  5018.4  1942.4  5039.3 1943.41  5051.7 1942.67
  5062.2 1943.17  5067.7 1944.15  5090.5 1942.64  5096.1 1943.53  5106.8 1943.99
  5141.8 1943.11  5159.1  1943.5  5272.3 1943.12  5347.6 1944.46  5353.1 1945.21
  5382.7 1944.23  5404.8 1944.77  5570.3 1945.04  5752.8 1947.41  5895.5 1947.14
  5918.3 1948.25  5969.6 1948.02  5986.9 1948.55  5992.4 1948.09  6006.5 1948.73
#Mann= 5 ,-1 , 0
  4143.1    .045       0  4277.2    .035       0  4722.6     .07       0
  5014.4     .07       0  5018.4     .07       0
Bank Sta=5014.4,5018.4
XS Rating Curve= 0 ,0
Exp/Cntr=0.3,0.1

Type RM Length L Ch R = 1 ,102006  ,466,466,466
BEGIN DESCRIPTION:
BULL WAGON CREEK 92.0
END DESCRIPTION:
XS GIS Cut Line= 3
      1516355.01        6825338.        1517355.        6825038.
      1517874.64      6824505.02
#Sta/Elev= 30
  3955.8 1948.29  4087.2  1946.8  4471.7 1942.11    4604 1941.71  4703.1 1939.69
  4708.4 1940.05  4769.3 1939.38  4780.6 1938.76    4885 1937.86    4945 1937.99
  4958.1 1938.49  4978.1 1937.56  4989.4 1938.35  5013.9 1937.96  5049.3 1938.46
  5141.2 1937.68  5176.6 1938.53  5195.8 1937.33    5196 1936.83  5199.5 1936.83
  5199.8 1937.33  5261.5 1938.58  5296.8 1938.36    5403 1939.34  5565.6 1943.23
  5650.4 1943.23  5657.4 1943.94  5692.9 1944.51  5721.2 1945.94  5744.2 1946.16
#Mann= 5 ,-1 , 0
  3955.8    .045       0  4087.2    .035       0  4471.7     .07       0
  5195.8     .07       0  5199.8     .07       0
Bank Sta=5195.8,5199.8
XS Rating Curve= 0 ,0
Exp/Cntr=0.3,0.1

Type RM Length L Ch R = 1 ,101540  ,411,411,411
BEGIN DESCRIPTION:
BULL WAGON CREEK 91.0
END DESCRIPTION:
XS GIS Cut Line= 3
      1517174.27      6825869.72      1517716.96      6825279.82
      1517954.99      6824838.02
#Sta/Elev= 30
  4209.3 1941.19    4237 1939.68  4295.8 1939.73  4317.4 1937.31  4486.9 1934.54
  4692.2 1934.59    4728 1933.58  4741.6 1930.28  4784.1 1933.79  4840.8 1934.03
  4862.4 1939.12  4881.4 1938.55  4940.1  1929.3  4980.6 1926.35  4980.8 1925.85
  4984.6 1926.35  4989.4  1927.7  5039.8 1926.48  5060.9 1929.76    5078 1934.85
  5115.2 1937.97  5137.9    1934    5172 1933.35  5187.5 1930.72  5209.4 1936.09
  5240.1 1937.85  5262.8 1934.12  5286.9 1934.89  5394.6 1938.28  5512.7 1941.45
#Mann= 8 ,-1 , 0
  4209.3    .035       0    4237     .07       0  4881.4    .035       0
  4980.6    .035       0  4984.6    .035       0  5060.9     .07       0
  5286.9     .16       0  5394.6     .07       0
Bank Sta=4980.6,4984.6
XS Rating Curve= 0 ,0
Exp/Cntr=0.3,0.1

Type RM Length L Ch R = 1 ,101129  ,228,228,228
BEGIN DESCRIPTION:
Mapping XS 4b90b977
END DESCRIPTION:
XS GIS Cut Line= 4
       1518038.2      6825422.29      1518004.82      6825340.11
      1517983.99      6825194.28      1518017.57      6825041.85
#Sta/Elev= 30
  4913.4 1937.24  4918.4 1937.24  4934.7 1934.63  4950.4 1928.87  4958.8 1926.95
  4964.2 1926.81    4970 1925.89  4970.3 1925.39  4973.8 1925.39    4974 1925.89
  4982.8 1926.28  4988.3 1927.08  4993.7 1926.52  5005.7 1926.35  5024.4 1930.07
  5037.9 1931.71  5044.6 1931.68  5064.8 1935.01  5095.1 1934.81  5108.6 1932.77
    5112 1932.73  5125.5 1932.34    5145 1933.24  5166.1 1933.45  5186.6 1934.51
  5196.8 1934.39    5207 1935.05  5237.7 1935.58    5289 1937.12  5305.5  1937.1
#Mann= 5 ,-1 , 0
  4913.4     .07       0    4970     .07       0    4974     .07       0
    5112     .16       0  5237.7     .07       0
Bank Sta=4970,4974
XS Rating Curve= 0 ,0
Exp/Cntr=0.3,0.1

Type RM Length L Ch R = 1 ,100901  ,266,266,266
BEGIN DESCRIPTION:
Mapping XS 81b19c78
END DESCRIPTION:
XS GIS Cut Line= 3
      1518241.13      6825320.87      1518210.55       6825269.8
      1518176.69      6825027.58
#Sta/Elev= 30
  4948.6 1936.51  4954.3 1936.44  4963.6 1934.93  4969.9 1934.44  4985.4 1928.19
  4991.2 1927.13  4996.6  1925.5  4996.8    1925  5000.3    1925  5000.6  1925.5
  5013.5 1926.18  5019.4 1926.01  5030.1 1925.62  5040.2 1926.03  5050.3 1929.72
  5060.4 1934.52  5070.5 1935.82    5085  1935.9  5090.7  1936.3  5100.8 1936.39
    5121 1937.11  5141.2 1937.12  5156.5 1937.64  5161.5 1937.32  5171.5 1937.45
  5181.6 1938.02  5201.8 1938.37  5227.9 1939.22    5233 1938.94  5252.7 1939.71
#Mann= 4 ,-1 , 0
  4948.6     .07       0  4996.6     .07       0  5000.6     .07       0
  5019.4     .16       0
Bank Sta=4996.6,5000.6
XS Rating Curve= 0 ,0
Exp/Cntr=0.3,0.1

Type RM Length L Ch R = 1 ,100635  ,305,305,305
BEGIN DESCRIPTION:
Mapping XS a4d1797f
END DESCRIPTION:
XS GIS Cut Line= 3
      1518478.34      6825205.71      1518434.51       6825144.8
      1518325.14      6824957.31
#Sta/Elev= 30
  4935.3 1935.05  4944.1 1935.84  4950.3 1935.97    4965 1931.66  4971.1 1928.88
  4977.7 1923.71    4978 1923.21  4981.5 1923.21  4981.7 1923.71  4985.9 1924.36
    4989 1924.26  4994.1  1924.1  5000.6 1924.43  5006.2 1925.53  5010.3 1925.53
  5015.9 1931.75  5021.6  1933.3  5029.8 1939.69  5080.4 1940.37  5096.1 1940.26
  5101.9 1940.96  5117.6 1940.92  5133.3 1941.38  5139.1 1941.37    5155 1940.27
  5160.6 1940.51  5168.7 1939.99  5198.2  1939.3  5203.6 1939.85  5227.4 1939.83
#Mann= 7 ,-1 , 0
  4935.3     .07       0  4977.7     .07       0  4981.7     .07       0
    4989     .16       0  5006.2     .07       0    5155    .035       0
  5198.2     .07       0
Bank Sta=4977.7,4981.7
XS Rating Curve= 0 ,0
Exp/Cntr=0.3,0.1

Type RM Length L Ch R = 1 ,100330  ,251,251,251
BEGIN DESCRIPTION:
Mapping XS d34debeb
END DESCRIPTION:
XS GIS Cut Line= 3
      1518723.94      6825054.79      1518690.87      6824999.84
      1518412.92       6824869.8
#Sta/Elev= 30
  4937.4 1935.16  4942.3 1935.28    4957 1932.56  4963.6 1930.26  4969.5 1929.14
  4979.2  1926.3    4985 1923.93  4997.7 1923.13  4997.9 1922.63  5001.4 1922.63
  5001.7 1923.13  5021.1 1925.02  5030.1 1928.22  5038.4 1929.42    5044 1931.64
  5054.1 1931.97  5118.4 1932.64  5135.3  1933.5  5140.8 1933.15  5158.2 1933.78
  5163.7 1933.33    5181  1934.1  5186.5 1933.66  5203.8 1934.83  5209.4 1933.91
  5226.7 1934.98  5232.2 1934.36  5276.7 1935.29  5295.1 1936.26  5308.4 1935.89
#Mann= 5 ,-1 , 0
  4937.4     .07       0  4997.7     .07       0  5001.7     .07       0
  5054.1     .16       0  5276.7     .07       0
Bank Sta=4997.7,5001.7
XS Rating Curve= 0 ,0
Exp/Cntr=0.3,0.1

Type RM Length L Ch R = 1 ,100079  ,348,348,348
BEGIN DESCRIPTION:
Mapping XS c046702d
END DESCRIPTION:
XS GIS Cut Line= 3
      1518931.29      6824929.02      1518907.89      6824897.84
      1518375.54      6824372.22
#Sta/Elev= 30
  4952.1 1934.87  4971.5 1930.82  4986.1 1924.03  4987.3 1921.56  4987.6 1921.06
  4991.3 1921.56  4992.7 1921.56  5014.2  1922.6  5035.5 1925.55  5042.5 1924.54
  5063.8 1925.65  5155.6 1925.23  5162.8 1926.23  5191.1 1925.56  5198.1 1924.38
  5205.2 1926.15  5212.2 1923.93  5219.3 1924.85  5226.4 1923.86  5233.5 1925.41
  5325.4  1927.3  5346.5 1925.11  5353.7 1927.51  5360.7 1926.75  5502.1    1930
  5537.5 1929.96  5558.7 1928.22  5572.8 1928.29  5622.4 1930.35  5739.2 1933.18
#Mann= 4 ,-1 , 0
  4952.1     .07       0  4987.3     .07       0  4991.3     .07       0
  4992.7     .16       0
Bank Sta=4987.3,4991.3
XS Rating Curve= 0 ,0
Exp/Cntr=0.3,0.1

Type RM Length L Ch R = 1 ,99731   ,505,505,505
BEGIN DESCRIPTION:
Mapping XS 850bba03
END DESCRIPTION:
XS GIS Cut Line= 3
      1518539.48      6825217.77      1519184.25      6824865.43
      1519675.99      6824574.92
#Sta/Elev= 30
  4266.8  1936.3  4315.7 1935.15  4321.4 1936.86  4337.5 1936.51  4343.2 1938.45
  4359.4 1936.39  4365.1 1938.52    4387 1937.45  4397.3    1935    4403 1936.68
  4419.1 1933.56  4462.8 1929.62  4683.3 1923.37  4718.9 1923.02  4735.1 1924.56
  4740.8 1922.47  4816.7 1922.52  4838.5 1920.83  4860.3 1922.44  4944.6 1922.27
  5037.1 1919.76  5041.6 1919.03  5042.1 1918.53  5047.1 1919.03  5050.2    1921
  5060.4 1920.18  5072.1 1922.85  5159.9 1924.42  5305.7 1929.07  5572.7 1933.31
#Mann= 7 ,-1 , 0
  4266.8     .07       0  4944.6     .16       0  5037.1     .07       0
  5041.6     .07       0  5047.1     .07       0  5060.4     .16       0
  5159.9     .07       0
Bank Sta=5041.6,5047.1
XS Rating Curve= 0 ,0
Exp/Cntr=0.3,0.1

Type RM Length L Ch R = 1 ,99226   ,390,390,390
BEGIN DESCRIPTION:
Mapping XS a4fb28b0
END DESCRIPTION:
XS GIS Cut Line= 4
      1518785.03      6825342.85      1519502.94      6825143.28
      1519581.07      6825058.65      1519650.27        6824877.
#Sta/Elev= 30
  4249.1 1928.73  4398.7 1925.96  4425.5  1924.7  4560.4 1923.57  4659.2 1921.85
    4685 1921.97  4693.4  1921.4  4726.5 1921.63  4732.8 1920.93  4767.1  1920.9
  4772.2 1920.24  4806.5 1920.46  4845.9 1919.66  4851.1  1920.1  4924.8 1918.58
    4959 1918.84  4975.6  1918.4  4992.7 1917.31  5077.3 1917.76  5098.3 1917.42
  5105.9 1916.16  5106.3 1915.66  5110.9 1915.66  5111.4 1916.16  5120.8 1916.49
  5135.7 1917.99  5142.2 1921.16  5152.9 1922.57  5241.3 1924.69  5303.8 1926.19
#Mann= 4 ,-1 , 0
  4249.1     .07       0  5105.9     .07       0  5111.4     .07       0
  5241.3    .035       0
Bank Sta=5105.9,5111.4
XS Rating Curve= 0 ,0
Exp/Cntr=0.3,0.1

Type RM Length L Ch R = 1 ,98836   ,682,682,682
BEGIN DESCRIPTION:
Mapping XS 70573959
END DESCRIPTION:
XS GIS Cut Line= 4
      1519048.77      6825578.11      1519548.51      6825438.42
      1519693.91      6825336.43      1519843.33      6825182.68
#Sta/Elev= 30
  4405.9 1921.78  4607.5 1919.31  4703.1 1919.19  4720.4 1918.59  4793.9  1918.3
  4799.1 1917.89  4833.2 1917.78  4838.4 1918.38  4858.9 1917.65  4951.4 1917.27
  4972.3 1917.54    4981 1916.01  4987.1 1914.14  4993.8 1912.78  4999.1 1912.63
  4999.6 1912.13  5004.3 1912.13  5004.7 1912.63  5016.7 1913.33  5030.4 1916.43
  5037.6 1916.93  5058.6 1916.12  5104.8 1916.84  5109.2 1917.49  5116.1  1917.6
  5137.5 1919.88  5151.6 1920.38  5208.2 1920.26  5249.5 1921.23  5316.8 1921.84
#Mann= 4 ,-1 , 0
  4405.9     .07       0  4999.1     .07       0  5004.7     .07       0
  5249.5    .035       0
Bank Sta=4999.1,5004.7
XS Rating Curve= 0 ,0
Exp/Cntr=0.3,0.1

Type RM Length L Ch R = 1 ,98154   ,191,191,191
BEGIN DESCRIPTION:
Mapping XS cad9330c
END DESCRIPTION:
XS GIS Cut Line= 4
      1518968.61      6826175.42      1519453.03      6825982.69
      1519708.24      6825727.48       1519812.4      6825266.57
#Sta/Elev= 30
  4410.7    1917  4635.9 1917.12  4751.2 1914.82  4822.1 1910.84  4905.7 1910.48
  4920.6 1907.66  4921.1 1907.16  4926.2 1907.66    4930 1909.79  4943.8 1911.61
  5042.8 1910.12    5064 1912.62  5078.2 1909.42  5147.9  1911.8  5233.7  1913.4
    5255 1912.09    5262 1913.44  5269.1 1911.42  5276.2 1913.64  5283.2  1912.2
  5289.1 1914.99  5299.3 1915.53  5312.9 1914.84  5333.4 1910.91  5390.8 1911.16
  5395.9 1912.78    5434 1910.88  5507.7 1912.14  5530.6 1917.25  5765.5  1920.9
#Mann= 4 ,-1 , 0
  4410.7     .07       0  4920.6     .07       0  4926.2     .07       0
  5147.9    .035       0
#XS Ineff= 2 , 0
       0                    5064       0 1912.62
Permanent Ineff=
       F       F
Bank Sta=4920.6,4926.2
XS Rating Curve= 0 ,0
Exp/Cntr=0.3,0.1

Type RM Length L Ch R = 1 ,97963   ,262,262,262
BEGIN DESCRIPTION:
Mapping XS 3b10a16f
END DESCRIPTION:
XS GIS Cut Line= 3
      1519333.23       6827230.1      1519637.92      6826066.03
        1519838.      6825281.32
#Sta/Elev= 30
  3800.6 1916.28  3999.2 1915.91  4050.9 1917.24  4186.6 1914.64  4216.2 1913.11
  4247.3 1906.92  4358.2 1905.45  4358.6 1904.95  4363.8 1905.45  4557.4 1909.19
  4764.1 1909.37  4784.8 1906.76  4835.7 1908.92  4852.2 1908.54  5003.9 1909.55
  5105.1 1912.91  5132.3  1909.1  5137.4 1911.44  5173.2 1907.62  5178.3    1909
  5249.5 1907.53  5336.7 1911.72  5377.6 1916.44  5413.3 1911.17  5418.4 1914.08
  5459.3 1916.46    5495 1911.74  5535.9 1912.53  5590.1 1918.15  5813.7 1920.85
#Mann= 5 ,-1 , 0
  3800.6    .035       0  4358.2    .035       0  4363.8    .035       0
  4835.7     .07       0  4852.2    .035       0
#XS Ineff= 2 , 0
       0                  4691.4       0 1909.86
Permanent Ineff=
       F       F
Bank Sta=4358.2,4363.8
XS Rating Curve= 0 ,0
Exp/Cntr=0.3,0.1

Type RM Length L Ch R = 1 ,97701   ,766,766,766
BEGIN DESCRIPTION:
Mapping XS 66733c88
END DESCRIPTION:
XS GIS Cut Line= 3
      1519455.63      6827266.57      1519716.05      6826318.63
      1519882.56      6825452.24
#Sta/Elev= 30
  3999.8  1914.2  4031.8 1914.34  4049.5  1915.4  4070.9  1913.8  4164.8 1913.18
  4265.6  1912.9  4366.4 1910.25  4430.1 1910.05  4435.3 1908.34  4444.2 1908.97
  4464.5 1906.86    4568 1905.83  4638.5  1905.4  4638.9  1904.9  4644.1  1905.4
  4668.8 1906.34  4838.3 1908.41  4845.1 1908.39  4850.3 1905.56  4864.7  1906.2
  4890.2  1908.5  4985.7 1908.07  5053.2 1905.75  5075.1 1907.54  5162.2 1907.31
  5167.3 1908.73  5214.2 1910.76  5238.1 1913.31  5537.4 1916.69  5865.1 1920.26
#Mann= 11 ,-1 , 0
  3999.8    .035       0  4031.8     .07       0  4164.8    .035       0
  4265.6     .07       0  4366.4    .035       0    4568     .07       0
  4638.5     .07       0  4644.1     .07       0  4668.8    .035       0
  4864.7     .07       0  5537.4    .035       0
Bank Sta=4638.5,4644.1
XS Rating Curve= 0 ,0
Exp/Cntr=0.3,0.1

Type RM Length L Ch R = 1 ,96935   ,690,690,690
BEGIN DESCRIPTION:
Mapping XS 89af4706
END DESCRIPTION:
XS GIS Cut Line= 3
      1519517.28      6827316.88      1520090.18      6826876.79
      1520259.45      6826186.67
#Sta/Elev= 30
  4274.9 1913.04  4308.8 1913.03  4410.7 1910.21  4493.7 1907.72  4549.8 1907.15
  4572.6    1906  4686.8 1904.27  4814.3 1903.67  4842.6 1902.24  4857.1 1903.23
  4900.6 1903.73  4918.6 1901.74  4919.1 1901.24  4924.3 1901.74  4927.8 1903.25
  4940.7 1902.95  4971.3 1902.97  4985.8 1901.93    5007 1902.29  5082.1 1902.62
  5088.7 1903.27  5123.6 1903.22  5160.1 1904.18  5278.8 1904.12  5285.5 1904.14
  5366.8 1904.82  5438.8 1907.79  5490.3 1907.97  5562.4  1909.8  5707.9 1911.46
#Mann= 8 ,-1 , 0
  4274.9     .16       0  4410.7     .07       0  4918.6    .035       0
  4924.3     .07       0  4940.7    .035       0    5007     .07       0
  5278.8    .035       0  5285.5     .07       0
Bank Sta=4918.6,4924.3
XS Rating Curve= 0 ,0
Exp/Cntr=0.3,0.1

Type RM Length L Ch R = 1 ,96245   ,555,555,555
BEGIN DESCRIPTION:
Mapping XS fec62ec7
END DESCRIPTION:
XS GIS Cut Line= 3
      1519535.52        6827382.       1520540.7      6827290.85
      1520905.27      6827113.78
#Sta/Elev= 30
  3974.2 1912.76  4128.1 1910.05  4204.6 1908.36  4292.6 1902.61  4395.4  1900.7
  4455.6 1900.27  4485.8 1901.12    4536 1901.11  4576.1 1899.63  4616.3 1900.43
  4629.4 1899.52  4666.5 1898.93  4756.9 1899.44  4850.6 1898.84  4867.3 1899.56
  4877.4 1898.77  4937.6  1898.2  5010.5 1898.63    5021 1897.92  5021.5 1897.42
  5030.5 1897.92    5047 1901.01    5055 1902.83  5065.3 1904.04  5070.9 1903.75
  5087.9 1906.26  5093.5 1905.66  5110.5 1907.36  5241.7 1908.02  5388.8 1909.29
#Mann= 6 ,-1 , 0
  3974.2     .16       0  4128.1     .07       0    5021     .07       0
  5030.5     .07       0    5047    .035       0  5241.7    .045       0
Bank Sta=5021,5030.5
XS Rating Curve= 0 ,0
Exp/Cntr=0.3,0.1

Type RM Length L Ch R = 1 ,95690   ,186,186,186
BEGIN DESCRIPTION:
Mapping XS ba55cdc2
END DESCRIPTION:
XS GIS Cut Line= 3
      1519525.05       6827452.3      1520374.03      6827642.42
      1521084.85      6827783.02
#Sta/Elev= 30
  4149.4 1912.52  4158.3 1912.44  4364.6 1909.31  4374.8 1908.43  4380.7 1906.45
  4385.8 1907.83  4397.5 1905.06  4405.5 1903.57    4424 1902.72  4456.8 1903.08
  4497.8 1900.86    4590 1899.04  4723.2 1899.88  4791.6 1898.24  4799.4 1898.81
  4825.7 1899.03  4834.9 1897.22  4840.1 1898.02  4856.4 1896.62  4876.9  1898.4
  4994.9 1896.34  4995.4 1895.84  5004.9 1896.34    5051 1897.92  5126.5 1898.18
  5153.2  1899.5    5265 1903.04  5590.6 1905.78  5703.4 1906.07    5744 1907.17
#Mann= 8 ,-1 , 0
  4149.4    .035       0  4158.3     .16       0  4397.5    .035       0
  4799.4     .07       0  4994.9     .07       0  5004.9     .07       0
  5153.2    .035       0  5590.6    .045       0
Bank Sta=4994.9,5004.9
XS Rating Curve= 0 ,0
Exp/Cntr=0.3,0.1

Type RM Length L Ch R = 1 ,95504   ,965,965,965
BEGIN DESCRIPTION:
Mapping XS 8f4c5ccf
END DESCRIPTION:
XS GIS Cut Line= 3
      1519376.64      6827618.98      1520345.39       6827822.1
      1521144.85      6828004.39
#Sta/Elev= 30
  4000.3  1911.9  4059.9 1909.76    4111 1909.77  4178.7 1908.53  4233.6 1907.99
  4254.1 1907.25  4284.7 1904.81  4361.2  1903.6    4406 1902.16  4455.9 1899.32
  4555.7  1897.1  4662.8 1896.14  4744.5 1897.67  4785.4 1896.89  4887.5 1897.67
    5000 1896.62  5005.2 1895.01  5005.7 1894.51  5015.3 1895.01  5030.7 1896.51
  5071.8 1896.07  5080.5 1897.12  5085.6 1896.33  5112.8 1895.66  5133.8 1896.59
  5191.6 1901.86  5297.4 1901.81  5512.8 1904.07  5579.2 1903.89  5810.1 1905.84
#Mann= 5 ,-1 , 0
  4000.3    .045       0  4178.7     .07       0  5005.2     .07       0
  5015.3     .07       0  5191.6    .035       0
Bank Sta=5005.2,5015.3
XS Rating Curve= 0 ,0
Exp/Cntr=0.3,0.1

Type RM Length L Ch R = 1 ,94539   ,1007,1007,1007
BEGIN DESCRIPTION:
Mapping XS 41bbf3cb
END DESCRIPTION:
XS GIS Cut Line= 4
       1519321.5      6828039.55      1519929.16      6828187.12
      1520324.12      6828282.61      1521257.32      6828291.29
#Sta/Elev= 30
  4400.4 1908.51  4421.8 1909.49  4453.9  1907.1  4495.6 1906.38  4517.2 1907.77
  4537.4 1905.79  4568.6 1904.89  4609.8 1906.16  4631.2 1904.08  4655.8 1903.49
    4667 1903.21    4723 1904.29  4751.4 1902.13  4815.6 1901.32  4840.1 1902.26
  4857.5 1900.64    4898 1899.56  4959.7 1900.41  4970.5  1899.1  4995.8 1889.56
  4996.3 1889.06    5006 1889.56  5007.1 1892.01  5054.1 1893.29  5206.6 1893.03
  5258.1 1894.86  5394.1  1894.7  5813.6 1900.32    5983 1901.03  6365.3 1906.15
#Mann= 8 ,-1 , 0
  4400.4     .07       0  4421.8    .045       0  4655.8     .07       0
    4667    .045       0  4857.5     .07       0  4995.8     .07       0
    5006     .07       0  5813.6    .035       0
Bank Sta=4995.8,5006
XS Rating Curve= 0 ,0
Exp/Cntr=0.3,0.1

Type RM Length L Ch R = 1 ,93532   ,563,563,563
BEGIN DESCRIPTION:
Mapping XS f5e458b2
END DESCRIPTION:
XS GIS Cut Line= 3
      1519356.26      6828829.48      1520406.59       6828755.7
      1521021.42      6828534.88
#Sta/Elev= 30
  3948.8 1901.49  3967.6 1902.14  3997.7 1900.47  4152.3 1898.88  4168.1 1898.55
  4210.8 1899.81  4228.2 1898.32  4255.1 1897.89  4408.7 1896.15  4428.7 1897.33
  4448.8 1895.47  4661.9 1893.39  4759.7 1892.11  4809.7 1892.61  4859.8 1891.37
  4879.8 1890.23  4909.9 1890.77    4940 1890.23  4961.7 1888.99  4990.1 1886.84
  4993.2 1886.09  4993.7 1885.59  5003.1 1885.59  5003.6 1886.09  5013.8 1888.43
  5021.3 1891.29  5053.2 1894.38  5112.8 1893.92  5273.5 1895.04    5655 1901.42
#Mann= 10 ,-1 , 0
  3948.8     .07       0  4152.3    .045       0  4210.8     .07       0
  4255.1    .045       0  4661.9     .07       0  4961.7    .045       0
  4993.2    .045       0  5003.6    .045       0  5013.8     .07       0
  5112.8    .035       0
Bank Sta=4993.2,5003.6
XS Rating Curve= 0 ,0
Exp/Cntr=0.3,0.1

Type RM Length L Ch R = 1 ,92969   ,965,965,965
BEGIN DESCRIPTION:
Mapping XS 1f3b3827
END DESCRIPTION:
XS GIS Cut Line= 3
       1519619.3      6829332.95      1520296.34      6829232.26
      1521067.15      6828947.55
#Sta/Elev= 30
  4306.1  1896.9    4322 1896.57  4342.2 1898.19  4370.6 1895.94  4490.4 1892.97
  4544.4 1892.43  4584.8 1892.77  4666.9 1891.78  4948.8 1891.03  4958.9 1890.05
    4969 1887.33  4973.9 1884.15  4974.4 1883.65  4983.9 1883.65  4984.4 1884.15
  4984.9 1884.82  4988.1 1885.76  5016.6 1887.47  5026.7 1887.44  5170.4 1888.62
  5224.2 1887.28  5243.9 1887.39  5255.7 1888.26  5279.7  1891.4  5310.1  1891.8
  5372.9 1894.41  5404.9 1894.13  5632.9 1897.23  5641.9 1897.25  5812.3  1900.1
#Mann= 8 ,-1 , 0
  4306.1    .045       0  4490.4     .07       0  4666.9    .045       0
  4973.9    .045       0  4984.4    .045       0  5026.7     .07       0
  5632.9    .045       0  5641.9    .035       0
Bank Sta=4973.9,4984.4
XS Rating Curve= 0 ,0
Exp/Cntr=0.3,0.1

Type RM Length L Ch R = 1 ,92004   ,454,454,454
BEGIN DESCRIPTION:
Mapping XS cf8c7165
END DESCRIPTION:
XS GIS Cut Line= 3
      1519694.75      6829824.28      1520170.47      6829740.94
      1521090.31      6829428.54
#Sta/Elev= 30
  4525.9 1897.19  4545.8 1896.87  4597.2 1895.96  4617.5 1897.35  4646.1 1894.47
  4728.8  1893.3  4781.4 1893.57  4901.8 1890.65  4938.1 1887.94  4997.6 1886.35
  5008.6 1882.74  5013.9 1882.74  5018.6 1879.92  5019.1 1879.42  5029.8 1879.92
  5036.8 1882.21  5045.3 1883.19  5068.2 1882.56  5125.7 1884.89  5256.5 1886.84
  5267.1 1886.03  5282.6 1886.96  5345.4 1886.47  5393.8 1888.37  5552.3 1891.58
  5747.2 1892.52  5858.5 1894.75  5890.2 1896.73  5906.4 1896.31  5980.3 1896.89
#Mann= 8 ,-1 , 0
  4525.9    .045       0  4545.8     .07       0  4728.8    .045       0
  4781.4     .07       0  5018.6     .07       0  5029.8     .07       0
  5747.2    .035       0  5906.4     .07       0
Bank Sta=5018.6,5029.8
XS Rating Curve= 0 ,0
Exp/Cntr=0.3,0.1

Type RM Length L Ch R = 1 ,91550   ,1337,1337,1337
BEGIN DESCRIPTION:
BULL WAGON CREEK 74.0
END DESCRIPTION:
XS GIS Cut Line= 3
      1519805.02        6829938.        1520455.        6830038.
      1521254.98      6829538.01
#Sta/Elev= 30
  4347.3 1896.84  4376.4 1893.96  4488.9 1894.15  4519.3 1891.72  4600.2 1888.34
  4639.4 1885.32  4644.5 1882.92  4681.2  1883.3  4701.4 1885.03  4762.1 1882.14
  4893.6 1883.85  4944.2 1882.19  4954.5 1882.89  4984.7 1881.72  4989.2 1878.51
  4989.7 1878.01  5000.4 1878.51  5002.4 1881.12  5019.7 1882.65  5049.1 1883.17
  5085.7 1888.08  5091.6 1886.96  5143.5 1886.89  5185.9 1887.23  5201.3 1888.43
  5389.9 1888.72  5563.3 1891.87  5578.6 1893.29  5746.1 1894.26  5948.3 1898.97
#Mann= 5 ,-1 , 0
  4347.3     .07       0  4954.5     .16       0  4989.2     .07       0
  5000.4     .16       0  5019.7     .07       0
Bank Sta=4989.2,5000.4
XS Rating Curve= 0 ,0
Exp/Cntr=0.3,0.1

Type RM Length L Ch R = 1 ,90213   ,432,432,432
BEGIN DESCRIPTION:
BULL WAGON CREEK 73.0
END DESCRIPTION:
XS GIS Cut Line= 3
      1519954.97      6830638.01        1520305.        6830538.
        1520955.        6829788.
#Sta/Elev= 30
  4630.9 1892.78  4641.3 1893.48  4662.1 1891.38  4714.1 1889.75  4766.1 1889.58
  4798.6 1891.19  4841.8 1889.18  4890.9 1884.51  4905.2 1885.06  4911.7 1882.65
  4922.1 1880.99    4939 1880.48  4967.2 1876.17  4967.7 1875.67  4978.4 1876.17
  4997.6 1877.39  5008.7 1878.36  5030.6 1876.82  5059.1 1879.21  5065.7 1878.43
  5151.2 1880.07  5186.3 1883.17  5264.2 1885.47    5626 1886.52  5902.4 1890.45
  5930.9 1892.14  5937.5 1894.48  5951.8 1894.35    5966 1892.56  5987.4 1892.93
#Mann= 5 ,-1 , 0
  4630.9     .07       0  4841.8     .16       0  4967.2     .07       0
  4978.4     .16       0  4997.6     .07       0
Bank Sta=4967.2,4978.4
XS Rating Curve= 0 ,0
Exp/Cntr=0.3,0.1

Type RM Length L Ch R = 1 ,89781   ,423,423,423
BEGIN DESCRIPTION:
BULL WAGON CREEK 72.0
END DESCRIPTION:
XS GIS Cut Line= 3
      1519851.87      6831031.58        1520605.        6830688.
      1521265.06      6830014.24
#Sta/Elev= 30
  4171.5 1896.68  4175.3 1896.68  4249.6  1895.8  4266.4 1896.62  4295.8 1893.22
  4328.8  1892.1  4357.9  1892.6  4427.7 1889.43  4651.5 1887.64  4693.1 1885.45
  4766.7 1882.88  4841.3 1877.55    4962 1878.41  5002.8 1876.87  5014.9 1874.67
  5015.4 1874.17  5026.2 1874.67  5048.8 1879.63  5084.1 1883.01  5102.2 1882.61
  5218.5 1884.57  5409.4 1884.68  5451.8 1886.88    5558 1886.78    5664 1889.97
  5755.9 1889.64  5826.6 1892.58  5840.7 1891.55  5847.9 1893.33  5942.5 1893.94
#Mann= 8 ,-1 , 0
  4171.5    .045       0  4175.3     .07       0  4249.6    .045       0
  4357.9     .07       0  4693.1     .16       0  5014.9     .07       0
  5026.2     .16       0  5102.2     .07       0
Bank Sta=5014.9,5026.2
XS Rating Curve= 0 ,0
Exp/Cntr=0.3,0.1

Type RM Length L Ch R = 1 ,89358   ,447,447,447
BEGIN DESCRIPTION:
Mapping XS ef59eebf
END DESCRIPTION:
XS GIS Cut Line= 4
        1520101.       6831536.8        1520542.      6831088.86
      1520969.09      6830418.72      1521270.56      6830117.25
#Sta/Elev= 30
  4325.3 1884.98  4345.6 1884.98  4465.7 1885.84    4685 1885.26  4928.3  1884.9
  4949.6 1883.39  4952.5 1879.93  4964.8 1878.33  4970.7 1874.66  4995.5 1873.19
    4996 1872.69  5006.9 1873.19  5014.2 1876.06  5022.4  1876.6  5101.1  1877.6
  5131.5 1881.59  5167.9 1883.05  5173.9 1880.84    5195  1879.3  5261.9 1878.73
  5392.2 1880.47  5428.6 1882.55  5476.9 1882.36  5507.3    1884  5652.9 1884.12
  5760.3 1887.14  5859.3 1886.57  5958.3 1889.87  6050.2 1889.31  6174.9 1892.44
#Mann= 6 ,-1 , 0
  4325.3    .045       0  4345.6     .07       0  4465.7    .045       0
    4685     .07       0  4995.5     .07       0  5006.9     .07       0
Bank Sta=4995.5,5006.9
XS Rating Curve= 0 ,0
Exp/Cntr=0.3,0.1

Type RM Length L Ch R = 1 ,88911   ,425,425,425
BEGIN DESCRIPTION:
Mapping XS 7c071df8
END DESCRIPTION:
XS GIS Cut Line= 4
      1520529.84      6831804.18      1520616.66      6831449.97
      1521196.52      6830925.66      1521480.64      6830454.44
#Sta/Elev= 30
  4209.3 1884.29  4415.3 1883.37    4525 1882.02  4595.6 1883.15  4659.2 1882.29
  4822.1    1875  4878.8 1874.64    4914 1875.53  4991.7 1874.64  4999.2 1872.49
  5007.6 1871.33  5008.1 1870.83  5019.1 1871.33  5034.3 1873.87  5041.7 1877.44
  5070.1 1878.55  5091.1 1877.49  5097.8 1878.38  5154.6 1879.34  5168.8 1880.92
  5303.3 1880.89  5360.7 1883.61  5477.2 1883.73  5550.9 1885.65  5578.1 1887.15
  5657.7 1886.48  5725.7 1888.21  5752.9 1889.73    5848 1889.63    5906 1891.68
#Mann= 5 ,-1 , 0
  4209.3     .07       0  4415.3    .035       0    4525     .07       0
  5007.6     .07       0  5019.1     .07       0
Bank Sta=5007.6,5019.1
XS Rating Curve= 0 ,0
Exp/Cntr=0.3,0.1

Type RM Length L Ch R = 1 ,88486   ,732,732,732
BEGIN DESCRIPTION:
Mapping XS 6a59b4ca
END DESCRIPTION:
XS GIS Cut Line= 4
      1520828.47      6831894.38      1521029.85      6831488.16
      1521272.91      6830956.91      1521536.79      6830526.36
#Sta/Elev= 30
  4565.7 1881.09  4646.1 1879.78  4746.8 1879.24  4944.8 1878.31  4963.5 1877.26
  4977.3 1872.69    4980 1869.72  4980.5 1869.22  4991.5 1869.72  4994.1  1871.1
  5008.1 1872.77  5039.6 1873.99  5173.2 1874.11  5206.2 1876.16  5250.2 1875.82
  5294.2 1878.01  5338.2 1878.54  5355.3 1879.83  5447.4 1881.09  5459.2 1882.48
  5492.1  1881.3  5550.4  1883.5  5691.7  1883.7    5771  1885.5  5801.4 1887.04
  5871.8 1886.53  5939.3 1888.07  5966.4  1889.6  6061.2 1889.31  6108.3 1890.54
#Mann= 6 ,-1 , 0
  4565.7    .035       0  4646.1     .07       0  4746.8    .035       0
  4944.8     .07       0    4980     .07       0  4991.5     .07       0
Bank Sta=4980,4991.5
XS Rating Curve= 0 ,0
Exp/Cntr=0.3,0.1

Type RM Length L Ch R = 1 ,87754   ,514,514,514
BEGIN DESCRIPTION:
Mapping XS fc80ae09
END DESCRIPTION:
XS GIS Cut Line= 3
      1521047.18      6831984.71      1521609.71      6831429.13
       1521849.3       6830918.7
#Sta/Elev= 30
  4219.1 1877.31  4397.2 1877.02  4573.2  1877.2    4689 1877.47  4717.3 1874.78
  4759.7 1872.97  4978.9 1871.09    4993 1870.57  4994.4 1868.21  4994.9 1867.71
  5005.5 1867.71    5006 1868.21  5018.2 1869.24  5030.8 1869.19  5053.6 1874.85
  5099.2 1876.27  5136.9 1878.84  5143.6    1879  5178.7 1882.98  5209.8 1887.94
  5247.1 1888.76  5269.9 1891.31  5292.8 1890.68  5331.3 1891.23  5366.7 1892.37
    5384 1892.12  5389.5  1893.2  5419.7 1891.99    5475 1892.76  5573.6 1892.77
#Mann= 7 ,-1 , 0
  4219.1     .07       0  4397.2    .035       0  4573.2     .07       0
  4994.4     .07       0    5006     .07       0  5018.2     .16       0
  5136.9     .07       0
Bank Sta=4994.4,5006
XS Rating Curve= 0 ,0
Exp/Cntr=0.3,0.1

Type RM Length L Ch R = 1 ,87240   ,565,565,565
BEGIN DESCRIPTION:
Mapping XS 1f472295
END DESCRIPTION:
XS GIS Cut Line= 4
      1521060.71      6832057.16      1521776.81      6831851.44
      1522011.19      6831729.05      1522203.68      6831302.44
#Sta/Elev= 30
  4150.5 1877.29  4394.3 1874.75  4545.1 1874.96  4617.4 1875.14  4676.5 1875.11
  4749.1 1868.48  4831.3 1869.98  4972.5 1870.34  4994.7 1865.33  4995.2 1864.83
  5006.3 1865.33  5016.9 1869.56  5022.5 1868.06  5028.9 1869.68  5044.6 1870.57
  5083.1 1870.42  5111.8  1872.5  5127.3 1873.43    5133 1875.74  5163.3 1879.56
  5202.6 1886.56    5216 1887.77  5306.1 1892.27  5345.5 1892.46  5427.2 1893.87
  5450.4    1893  5462.7 1894.32  5556.1 1897.72  5594.6 1896.68    5628 1897.75
#Mann= 8 ,-1 , 0
  4150.5     .07       0  4545.1    .035       0  4617.4     .07       0
  4994.7     .07       0  5006.3     .07       0  5111.8     .16       0
  5345.5     .07       0  5462.7    .035       0
Bank Sta=4994.7,5006.3
XS Rating Curve= 0 ,0
Exp/Cntr=0.3,0.1

Type RM Length L Ch R = 1 ,86675   ,574,574,574
BEGIN DESCRIPTION:
Mapping XS aea0a485
END DESCRIPTION:
XS GIS Cut Line= 3
      1521087.98       6832098.4      1522105.37      6832087.99
      1522789.43      6831844.92
#Sta/Elev= 30
  3708.2 1877.06  3904.4 1875.55    4125 1873.42    4323 1872.98  4527.3 1872.13
  4838.2 1870.78    4859  1870.2  4864.3 1870.74  4873.8 1869.71  4889.8 1869.56
  4895.1 1868.68  4977.1 1867.82  4990.6 1867.39  4992.6  1866.7  4995.4 1865.74
  4995.9 1865.24    5007 1865.74  5007.9 1866.58  5013.2 1866.88  5022.4 1869.36
    5033  1873.6  5038.8 1879.51  5044.1 1881.35  5054.2 1887.54  5064.3 1890.73
  5075.5 1892.77    5171 1893.13  5311.1 1895.24  5350.5  1894.6  5451.6 1895.33
#Mann= 10 ,-1 , 0
  3708.2    .035       0  3904.4     .07       0    4125    .035       0
    4323     .07       0  4527.3    .035       0  4838.2     .07       0
  4992.6     .16       0  4995.4     .07       0    5007     .16       0
  5350.5    .045       0
Bank Sta=4995.4,5007
XS Rating Curve= 0 ,0
Exp/Cntr=0.3,0.1

Type RM Length L Ch R = 1 ,86101   ,180,180,180
BEGIN DESCRIPTION:
Mapping XS e5870ce6
END DESCRIPTION:
XS GIS Cut Line= 2
      1521094.06      6832173.92      1522955.18        6832601.
#Sta/Elev= 30
  3706.4 1877.95  3719.1 1877.75  3841.9 1877.04  4021.9 1875.65  4058.5 1875.21
  4437.4 1872.08    4541 1871.52  4643.7 1870.51  4729.4 1868.19  4887.3 1867.25
    4918 1865.89  4954.1    1866  4969.3  1864.8  4989.9 1865.23  5004.5 1863.85
    5005 1863.35  5016.2 1863.85  5030.9 1866.77  5039.8 1867.03  5044.9 1868.54
  5082.2 1868.35  5143.8  1871.6  5178.7 1871.83  5256.6 1878.24  5355.3 1878.69
  5360.5 1880.45  5398.2 1884.03  5494.2 1885.21    5532 1886.68  5615.9 1887.22
#Mann= 9 ,-1 , 0
  3706.4     .07       0  3719.1    .035       0  3841.9     .07       0
  4021.9    .035       0  4058.5     .07       0  4437.4    .035       0
    4541     .07       0  5004.5     .07       0  5016.2     .07       0
Bank Sta=5004.5,5016.2
XS Rating Curve= 0 ,0
Exp/Cntr=0.3,0.1

Type RM Length L Ch R = 1 ,85921   ,677,677,677
BEGIN DESCRIPTION:
Mapping XS 1829363c
END DESCRIPTION:
XS GIS Cut Line= 3
      1520864.89      6832333.64      1522295.47      6832625.31
      1522958.69       6832778.1
#Sta/Elev= 30
  3530.3 1879.37  3561.4  1878.1    3907 1876.36  4072.3 1875.57  4103.9 1875.16
  4223.6 1874.75  4336.7 1872.77  4357.1 1873.56  4474.1 1870.88    4633 1869.79
  4669.9 1868.48  4744.9 1867.51  4773.7 1863.08  4774.2 1862.58  4785.4 1863.08
  4806.1 1868.44  4846.9 1865.67  4908.2 1865.54  4976.3 1867.14  5010.3 1863.22
  5041.1  1866.6  5115.9  1866.8  5205.1 1870.24  5377.8 1875.02  5382.9 1874.06
  5480.9 1876.43  5554.1 1880.75    5585 1880.43  5644.8 1883.59  5670.9 1883.47
#Mann= 12 ,-1 , 0
  3530.3     .07       0  3561.4    .035       0    3907     .07       0
  4072.3    .035       0  4103.9     .07       0  4474.1    .035       0
  4669.9     .07       0  4773.7    .035       0  4785.4     .07       0
  4976.3    .035       0  5205.1     .07       0  5480.9    .035       0
Bank Sta=4773.7,4785.4
XS Rating Curve= 0 ,0
Exp/Cntr=0.3,0.1

Type RM Length L Ch R = 1 ,85244   ,692,692,692
BEGIN DESCRIPTION:
Mapping XS 39309b9e
END DESCRIPTION:
XS GIS Cut Line= 4
      1521506.41      6832889.04      1522055.44      6833314.71
      1522268.04      6833251.55      1523054.41      6832847.28
#Sta/Elev= 30
  4083.5 1873.93  4127.8  1873.5  4295.4 1872.34  4349.7 1871.96  4664.1 1869.97
  4776.8 1868.85  4891.6 1869.32  4934.2 1868.66    4960 1867.15  4980.5 1860.21
    4981 1859.71  4992.3 1860.21  4996.4 1861.68  5007.8 1863.65  5043.9 1864.58
  5237.4 1863.84  5377.4  1865.4  5481.8 1866.89  5542.8 1866.79  5548.4 1867.49
  5609.3 1868.43    5648 1869.94    5698  1873.5  5736.8 1879.65  5758.9 1881.29
  5764.6 1880.31  5781.1 1881.34  5786.7 1880.87  5817.4 1882.07  5884.2 1882.82
#Mann= 11 ,-1 , 0
  4083.5    .035       0  4127.8     .07       0  4295.4    .035       0
  4349.7     .07       0  4664.1    .035       0  4891.6     .07       0
  4980.5     .07       0  4992.3     .07       0  4996.4     .07       0
  5237.4     .16       0  5377.4     .07       0
Bank Sta=4980.5,4992.3
XS Rating Curve= 0 ,0
Exp/Cntr=0.3,0.1

Type RM Length L Ch R = 1 ,84552   ,557,557,557
BEGIN DESCRIPTION:
Mapping XS 67e2a39c
END DESCRIPTION:
XS GIS Cut Line= 3
      1521860.87      6834661.47      1522785.32       6833463.6
      1523119.51      6832916.74
#Sta/Elev= 30
  3490.9 1871.37  3760.6 1868.92  3767.3 1868.11  3788.1 1869.11  3987.9 1868.66
  4373.3  1865.9  4537.2 1863.06  4672.2  1862.5  4686.7 1862.12  4694.8 1860.27
  4701.2 1860.98    4702 1858.63  4702.5 1858.13  4713.8 1858.63  4715.7 1862.82
  4771.8 1862.64  4836.1 1864.03  4881.6  1863.4  4949.1 1862.16  5014.7 1861.81
  5022.3 1858.88    5036 1862.09  5115.7 1862.76    5138 1863.55  5220.7 1864.33
  5373.5 1866.38  5457.9 1869.91  5510.1 1875.82    5538 1877.62  5644.9 1880.74
#Mann= 9 ,-1 , 0
  3490.9     .07       0    4702     .07       0  4713.8     .07       0
  4881.6     .16       0  4949.1     .07       0  5115.7     .16       0
    5138     .07       0  5220.7    .035       0  5373.5     .07       0
Bank Sta=4702,4713.8
XS Rating Curve= 0 ,0
Exp/Cntr=0.3,0.1

Type RM Length L Ch R = 1 ,83995   ,201,201,201
BEGIN DESCRIPTION:
Mapping XS f8bd3604
END DESCRIPTION:
XS GIS Cut Line= 3
      1522290.53      6835052.13      1523119.52      6833988.77
      1523249.48       6833001.1
#Sta/Elev= 30
  3499.2 1867.79  4008.4 1865.63  4090.3 1864.62  4266.9 1863.54  4293.7  1863.6
  4389.3 1863.46  4476.3 1862.21  4694.1 1859.49  4737.6 1860.32  4814.6 1860.04
    4907 1860.61  4959.2 1860.77  4969.3 1859.63  4979.4 1857.09  4989.5  1860.3
  5029.8  1861.1  5039.9 1859.61  5042.3 1856.44  5042.8 1855.94  5057.7 1856.44
  5060.1 1860.58  5070.2    1861  5251.7 1860.93  5271.9 1862.08  5483.7 1864.34
  5502.9 1865.17    5635  1866.8  5697.5 1868.58  5771.1 1871.66  5843.7  1876.9
#Mann= 12 ,-1 , 0
  3499.2     .07       0  4008.4    .035       0  4090.3     .07       0
  4266.9    .035       0  4293.7     .07       0  4476.3    .035       0
  4694.1     .07       0  4814.6     .16       0    4907     .07       0
  5042.3     .07       0  5057.7     .07       0  5502.9    .035       0
Bank Sta=5042.3,5057.7
XS Rating Curve= 0 ,0
Exp/Cntr=0.3,0.1

Type RM Length L Ch R = 1 ,83794   ,848,848,848
BEGIN DESCRIPTION:
Mapping XS ff9e7a17
END DESCRIPTION:
XS GIS Cut Line= 3
       1522959.8       6835310.8      1523319.17      6833914.98
      1523366.05      6833123.31
#Sta/Elev= 30
  3547.2 1863.69    3643 1863.37  3668.6 1864.15  3694.7 1863.56    3750 1863.98
  3766.9 1863.31  3790.7 1863.97  3849.5 1862.81  4088.2 1861.83  4500.1 1860.73
  4644.7 1858.64  4727.3 1859.51    4747 1860.29  4809.9 1859.61  4882.2 1860.37
  4902.8 1859.93  5001.5 1860.36  5017.9 1858.27  5018.4 1857.77  5032.8 1857.77
  5033.3 1858.27  5035.6 1860.22  5215.9 1860.59  5269.2 1861.41    5286 1861.46
  5454.1 1863.89  5546.5 1866.54  5636.7 1866.93  5736.8 1868.22  5781.6  1869.5
#Mann= 7 ,-1 , 0
  3547.2    .035       0  4088.2     .07       0  5017.9     .07       0
  5033.3     .07       0  5269.2    .035       0    5286     .07       0
  5454.1    .035       0
Bank Sta=5017.9,5033.3
XS Rating Curve= 0 ,0
Exp/Cntr=0.3,0.1

Type RM Length L Ch R = 1 ,82946   ,923,923,923
BEGIN DESCRIPTION:
Mapping XS 2618e492
END DESCRIPTION:
XS GIS Cut Line= 4
      1523069.15      6835357.73       1523959.8      6834128.53
      1524195.72       6833723.5      1523540.07      6832975.58
#Sta/Elev= 30
  3377.6 1862.67  4015.6 1860.22    4117 1859.61  4237.7 1857.71  4347.9 1855.34
  4374.2 1857.42  4384.2  1857.6    4405 1853.18  4405.8 1851.22  4406.3 1850.72
  4421.3 1851.22  4440.6 1856.73  4484.7 1857.54  4499.4  1860.2  4526.4 1857.31
    4627 1854.24  4656.3 1856.91  4979.2 1858.07  5000.7 1857.57  5023.5 1852.66
  5037.9 1857.44  5393.3  1861.6  5554.1 1862.14  5627.4 1862.49  5748.9 1863.59
  5895.1 1864.08    5944 1864.91  6022.7 1866.13  6286.7 1871.49  6358.9 1873.83
#Mann= 16 ,-1 , 0
  3377.6    .035       0  4015.6     .07       0    4117    .035       0
  4237.7     .07       0  4347.9    .035       0  4374.2     .07       0
  4405.8     .07       0  4421.3     .07       0  5393.3     .16       0
  5554.1     .07       0  5627.4     .16       0  5748.9     .07       0
  5895.1    .035       0    5944     .07       0  6022.7    .035       0
  6286.7     .07       0
Bank Sta=4405.8,4421.3
XS Rating Curve= 0 ,0
Exp/Cntr=0.3,0.1

Type RM Length L Ch R = 1 ,82023   ,652,652,652
BEGIN DESCRIPTION:
Mapping XS 581b28fc
END DESCRIPTION:
XS GIS Cut Line= 3
      1523095.23      6835487.89      1524043.13      6834597.28
       1525517.1      6834409.78
#Sta/Elev= 30
  3679.4 1862.26  3734.1 1862.31  3962.2 1862.34  4333.9  1859.2  4466.8 1858.39
  4499.1 1858.74  4648.2 1857.35  4798.5  1855.6  4832.1 1853.98  4853.6 1855.06
  4959.6 1855.86    4992 1855.23  5002.1  1853.6  5014.5 1853.33    5015 1852.83
    5030 1853.33  5062.6 1855.39  5133.1 1854.36  5223.9 1856.19  5350.3 1856.45
  5521.5 1856.61  5687.6 1857.92  5697.7 1857.04  5717.8 1858.46  5745.6 1858.44
    5810 1858.53  5869.5 1860.23  6071.7 1866.32  6252.1 1870.23  6465.9 1872.92
#Mann= 14 ,-1 , 0
  3679.4     .07       0  3734.1    .035       0  4333.9     .07       0
  4466.8    .035       0  4499.1     .07       0  4648.2    .035       0
  4798.5     .07       0  5014.5     .07       0    5030     .07       0
  5350.3    .035       0  5521.5     .07       0  5745.6    .035       0
  5869.5     .07       0  6071.7    .035       0
Bank Sta=5014.5,5030
XS Rating Curve= 0 ,0
Exp/Cntr=0.3,0.1

Type RM Length L Ch R = 1 ,81371   ,786,786,786
BEGIN DESCRIPTION:
Mapping XS d25d5729
END DESCRIPTION:
XS GIS Cut Line= 3
      1523199.35      6835581.67      1523827.85      6835076.44
      1525567.41      6834743.11
#Sta/Elev= 30
  3911.9 1862.25  4074.5 1861.94  4528.9 1858.06  4551.8 1857.95  4573.5 1857.22
  4586.4 1858.09    4677 1857.71  4925.3 1856.04  4980.1 1854.66  4995.9 1848.41
  4996.4 1847.91    5012 1848.41  5020.8 1853.95  5206.9 1853.91  5381.9 1854.33
  5499.4 1853.51  5519.8  1852.5  5540.1 1853.97  5698.6 1854.59  5706.2  1854.4
  5800.8 1854.78  5920.5 1857.48  6069.8 1864.12  6140.9 1865.44  6161.2 1867.23
  6191.8 1866.19  6232.5 1868.14  6307.5 1869.19  6408.8 1870.58  6489.5 1871.43
#Mann= 15 ,-1 , 0
  3911.9    .035       0  4528.9     .07       0  4551.8    .035       0
    4677     .07       0  4925.3    .035       0  4995.9    .035       0
    5012    .035       0  5206.9     .07       0  5381.9    .035       0
  5698.6     .07       0  5706.2    .035       0  5800.8     .07       0
  5920.5    .035       0  6307.5     .07       0  6408.8    .035       0
Bank Sta=4995.9,5012
XS Rating Curve= 0 ,0
Exp/Cntr=0.3,0.1

Type RM Length L Ch R = 1 ,80585   ,1794,1794,1794
BEGIN DESCRIPTION:
Mapping XS 48c88846
END DESCRIPTION:
XS GIS Cut Line= 3
       1523260.1      6835941.04      1523890.35      6835706.65
      1525800.92      6835238.12
#Sta/Elev= 30
  4300.4 1861.47  4448.2 1860.63  4767.4 1857.32  4815.7 1856.72  4959.1 1854.64
  4967.1 1853.95  4972.6 1852.24  4977.8 1852.24  4982.5 1848.67    4983 1848.17
  4998.8 1848.67  5018.8  1850.7  5049.7 1850.14  5073.8 1851.44  5156.9 1850.75
  5265.9 1851.61  5483.4 1851.17  5523.3 1851.73    5924 1852.35  5947.8 1852.25
  6191.2 1852.48  6357.3 1856.05  6378.4 1857.41  6398.5 1861.96    6406 1862.82
    6450 1864.63  6561.8 1866.33  6785.3 1870.15  6893.2 1871.89    6940 1872.89
#Mann= 16 ,-1 , 0
  4300.4     .07       0  4448.2    .035       0  4767.4     .07       0
  4815.7    .035       0  4959.1     .07       0  4982.5     .07       0
  4998.8     .07       0  5483.4     .16       0  5523.3     .07       0
    5924    .035       0  5947.8     .07       0  6191.2    .035       0
    6406     .07       0  6561.8    .035       0  6785.3     .07       0
  6893.2    .035       0
Bank Sta=4982.5,4998.8
XS Rating Curve= 0 ,0
Exp/Cntr=0.3,0.1

Type RM Length L Ch R = 1 ,78791   ,1227,1227,1227
BEGIN DESCRIPTION:
Mapping XS 0bfd67df
END DESCRIPTION:
XS GIS Cut Line= 3
      1523322.64      6836560.82      1523999.73      6836326.44
      1525930.98       6836191.1
#Sta/Elev= 30
  4289.5 1865.77  4865.8 1856.95  4923.2 1854.94  4937.5 1852.39  4948.1 1851.95
  4961.7 1847.91  4967.7 1846.97  4990.8  1844.6  5061.4 1845.71  5071.4 1846.12
  5101.5 1851.36  5121.6 1848.08  5171.7 1847.44  5372.2  1849.1  5552.6 1848.35
    5693 1846.76    5713 1844.73  5743.1 1844.89  5744.9 1843.61  5745.4 1843.11
  5761.3 1843.61  5763.1 1846.73  5774.3 1847.09    6104 1848.54  6244.3 1846.73
    6351 1850.46  6565.1 1856.18  6655.5 1856.98  6854.4 1859.33    6942 1860.26
#Mann= 9 ,-1 , 0
  4289.5    .035       0  4865.8     .07       0  4961.7    .035       0
  4967.7     .07       0  5744.9     .07       0  5761.3     .07       0
    6351    .035       0  6655.5     .07       0  6854.4    .035       0
#XS Ineff= 2 , 0
       0  5101.5 1851.36               0
Permanent Ineff=
       F       F
Bank Sta=5744.9,5761.3
XS Rating Curve= 0 ,0
Exp/Cntr=0.3,0.1
