--- MULBERRY CREEK TRIBUTARY 15.prj (project) ---

Proj Title=MULBERRY CREEK TRIBUTARY 15 Base Level Engineering
Current Plan=p01
Default Exp/Contr=0.3,0.1
English Units
Geom File=g01
Flow File=f01
Plan File=p01
Y Axis Title=Elevation
X Axis Title(PF)=Main Channel Distance
X Axis Title(XS)=Station
BEGIN DESCRIPTION:
MULBERRY CREEK TRIBUTARY 15
END DESCRIPTION:
DSS Export Rating Curves= 0
DSS Export Rating Curve Sorted= 0
DSS Export Volume Flow Curves= 0
DXF OffsetX= 0
DXF OffsetY= 0
DXF ScaleX= 1
DXF ScaleY= 10

--- MULBERRY CREEK TRIBUTARY 15.p01 (plan) ---

Plan Title=Multiple Run
Short Identifier=Multiple
Geom File=g01
Flow File=f01
Subcritical Flow
K Sum by GR= 0
Std Step Tol= 0.01
Critical Tol= 0.01
Num of Std Step Trials= 20
Max Error Tol= 0.3
Flow Tol Ratio= 0.001
Split Flow NTrial= 30
Split Flow Tol= 0.02
Split Flow Ratio= 0.02
Log Output Level= 0
Friction Slope Method= 1
Unsteady Friction Slope Method= 2
Unsteady Bridges Friction Slope Method= 1
Parabolic Critical Depth
Global Vel Dist=  1 , 1 , 1
Global Log Level= 0
CheckData=True
Encroach Param= -1, 0, 0, 0
BEGIN DESCRIPTION:
Multiple Run
END DESCRIPTION:

--- MULBERRY CREEK TRIBUTARY 15.f01 (steady flow) ---

Flow Title=Multiple
Program Version=4.10
Number of Profiles= 7
Profile Names=10-year,25-year,50-year,1pct_min,100-year,1pct_plu,500-year
River Rch & RM=MULBERRY CREEK T,Reach-1         ,42068
     166     224     271     163     326     650     477
River Rch & RM=MULBERRY CREEK T,Reach-1         ,34541
     262     364     447     274     547    1091     827
River Rch & RM=MULBERRY CREEK T,Reach-1         ,32681
     424     600     747     462     923    1841    1427
River Rch & RM=MULBERRY CREEK T,Reach-1         ,23123
     630     909    1147     719    1434    2861    2273
River Rch & RM=MULBERRY CREEK T,Reach-1         ,22747
     673     970    1224     766    1528    3049    2417
River Rch & RM=MULBERRY CREEK T,Reach-1         ,16709
     706    1019    1286     805    1607    3206    2544
River Rch & RM=MULBERRY CREEK T,Reach-1         ,14707
     763    1103    1394     874    1743    3478    2764
River Rch & RM=MULBERRY CREEK T,Reach-1         ,7261
     930    1353    1717    1080    2154    4299    3441
Boundary for River Rch & Prof#=MULBERRY CREEK T,Reach-1         , 1
Up Type= 0
Dn Type= 3
Dn Slope=0.00185
Boundary for River Rch & Prof#=MULBERRY CREEK T,Reach-1         , 2
Up Type= 0
Dn Type= 3
Dn Slope=0.00185
Boundary for River Rch & Prof#=MULBERRY CREEK T,Reach-1         , 3
Up Type= 0
Dn Type= 3
Dn Slope=0.00185
Boundary for River Rch & Prof#=MULBERRY CREEK T,Reach-1         , 4
Up Type= 0
Dn Type= 3
Dn Slope=0.00185
Boundary for River Rch & Prof#=MULBERRY CREEK T,Reach-1         , 5
Up Type= 0
Dn Type= 3
Dn Slope=0.00185
Boundary for River Rch & Prof#=MULBERRY CREEK T,Reach-1         , 6
Up Type= 0
Dn Type= 3
Dn Slope=0.00185
Boundary for River Rch & Prof#=MULBERRY CREEK T,Reach-1         , 7
Up Type= 0
Dn Type= 3
Dn Slope=0.00185
DSS Import GetInterval= 0
DSS Import GetPeak= 0
DSS Import FillOption= 0

--- MULBERRY CREEK TRIBUTARY 15.g01 (geometry) ---

Geom Title=Existing Conditions
Program Version=4.10

River Reach=MULBERRY CREEK T,Reach-1
Reach XY= 30
        1509905.        6853838.      1510894.49      6855777.53
      1511664.72      6855898.78      1513052.55      6857332.54
      1514520.22      6857837.48      1515253.37      6857641.13
      1516349.83      6858592.59      1516564.12      6860444.76
      1517399.56      6860393.17      1517598.79       6861580.2
      1518661.17      6861095.76      1521199.41      6863593.61
      1521311.05      6864136.42      1521858.41      6864230.62
      1522374.76      6863737.96      1523075.03      6864188.44
      1523665.45      6863738.53      1524861.66      6863896.98
      1525599.61      6864385.56        1525605.        6865388.
      1527207.55      6865692.98       1527510.9      6866386.03
       1528188.6      6866171.18        1528105.        6867588.
       1528594.9       6868027.7      1530403.35       6867591.1
      1530265.79      6868348.37      1531394.57      6869378.17
       1531345.3      6869777.84        1531755.        6869488.

Type RM Length L Ch R = 1 ,42068   ,583,583,583
BEGIN DESCRIPTION:
MULBERRY CREEK TRIBUTARY 15 44.0
END DESCRIPTION:
XS GIS Cut Line= 3
      1509205.04      6854137.99       1509978.4      6853911.31
        1510455.        6853538.
#Sta/Elev= 30
  4194.1  1846.5  4249.4 1845.03  4298.3 1844.28  4329.5  1844.4  4436.5  1842.3
  4475.4 1841.25  4498.9 1842.06  4604.3  1839.3  4633.8 1839.38  4671.1 1838.39
  4704.5 1838.19  4756.8 1838.85  4892.4 1838.43  5013.1 1836.85  5034.9 1836.48
    5041 1835.58  5041.3 1835.08  5044.8 1835.08    5045 1835.58  5063.8 1836.84
  5099.1 1837.65    5128 1837.57  5163.3 1839.22  5212.2  1840.2  5262.8 1841.47
  5320.6 1841.47  5405.6 1842.22    5449 1843.19  5544.5 1843.49  5605.4 1844.11
#Mann= 8 ,-1 , 0
  4194.1    .045       0  4436.5     .07       0  4633.8    .045       0
  5013.1     .07       0    5041    .045       0    5045     .07       0
  5212.2    .035       0  5544.5     .07       0
Bank Sta=5041,5045
XS Rating Curve= 0 ,0
Exp/Cntr=0.3,0.1

Type RM Length L Ch R = 1 ,41485   ,590,590,590
BEGIN DESCRIPTION:
Mapping XS ac8a84b5
END DESCRIPTION:
XS GIS Cut Line= 3
      1509153.47      6854417.95      1510064.97      6854449.21
       1510647.5      6853882.27
#Sta/Elev= 30
  4052.4 1846.77    4114 1845.09  4225.6 1843.23  4258.3 1842.76  4284.1  1842.8
  4384.1 1840.63  4434.2 1840.34  4515.8 1838.25  4597.2 1836.91  4704.3  1835.8
  4744.3 1834.75  4786.3 1834.76  4832.8 1833.68  4894.4 1832.66  4924.4 1832.82
  4993.5 1831.73  4998.7 1831.22  4998.9 1830.72  5002.4 1830.72  5002.7 1831.22
  5021.8  1832.1  5063.5 1832.65  5156.3 1835.17  5184.6 1835.24    5234 1836.58
  5311.9 1837.48  5389.6 1839.21  5481.5 1839.95  5552.2 1841.33  5777.3 1842.95
#Mann= 9 ,-1 , 0
  4052.4    .045       0  4225.6     .07       0  4258.3    .045       0
  4515.8     .07       0  4597.2    .045       0  4832.8     .07       0
  4998.7     .07       0  5002.7     .07       0  5063.5    .045       0
Bank Sta=4998.7,5002.7
XS Rating Curve= 0 ,0
Exp/Cntr=0.3,0.1

Type RM Length L Ch R = 1 ,40895   ,502,502,502
BEGIN DESCRIPTION:
Mapping XS ced9f61c
END DESCRIPTION:
XS GIS Cut Line= 3
      1509106.65      6855048.16       1510273.3      6854970.04
      1510960.41       6854439.1
#Sta/Elev= 30
  3785.3 1843.17  3853.8 1841.81  3903.9 1841.63  3974.1 1839.78  4044.2 1839.73
  4144.4 1838.03  4204.6 1838.13  4264.7 1836.64  4324.9 1836.38  4364.9  1835.3
  4425.1 1834.98  4505.3 1833.29  4565.4 1833.09  4642.8 1831.53  4755.7 1830.77
    4836 1829.43  4896.1 1829.76  4936.2 1828.47  4985.4 1828.64  4991.5 1828.19
  4991.8 1827.69  4995.3 1827.69  4995.5 1828.19  5049.7 1829.62  5064.2 1828.99
  5143.6 1829.62  5491.6 1834.87  5634.7 1835.77  5719.8 1837.27  5822.9 1837.58
#Mann= 5 ,-1 , 0
  3785.3    .045       0  4642.8     .07       0  4991.5     .07       0
  4995.5     .07       0  5143.6    .045       0
Bank Sta=4991.5,4995.5
XS Rating Curve= 0 ,0
Exp/Cntr=0.3,0.1

Type RM Length L Ch R = 1 ,40393   ,607,607,607
BEGIN DESCRIPTION:
Mapping XS abe4a2aa
END DESCRIPTION:
XS GIS Cut Line= 3
      1509189.93      6855584.63      1510455.59      6855339.83
       1510960.4      6854647.68
#Sta/Elev= 30
  3710.6 1837.94  3771.8 1836.54    3838 1836.45  3875.4 1835.48  4046.1 1833.83
  4144.5 1833.28    4243  1831.4  4377.8 1831.19  4455.3 1829.61  4530.6 1829.01
  4558.9 1829.68  4591.7  1828.6  4735.2  1827.6  4834.3 1826.82  4846.3 1827.43
  4874.8 1826.65  4931.6  1826.8  5005.7 1825.25  5005.9 1824.75  5009.7 1825.25
    5037 1826.41  5093.4 1826.02  5179.2 1827.05  5208.5 1826.27  5365.3 1829.38
  5419.6 1829.54  5465.8 1830.07  5486.6 1831.02  5572.4  1831.3  5856.4 1835.37
#Mann= 7 ,-1 , 0
  3710.6    .045       0  4046.1     .07       0  4735.2     .16       0
  4834.3     .07       0  5005.7     .07       0  5009.7     .07       0
  5419.6    .045       0
Bank Sta=5005.7,5009.7
XS Rating Curve= 0 ,0
Exp/Cntr=0.3,0.1

Type RM Length L Ch R = 1 ,39786   ,1458,1458,1458
BEGIN DESCRIPTION:
Mapping XS 0c576f68
END DESCRIPTION:
XS GIS Cut Line= 3
      1509106.66      6855933.58      1510841.01      6855652.33
        1511991.      6854944.65
#Sta/Elev= 30
    3222 1835.59    3232 1835.42  3392.5 1833.11  3574.9  1832.7  3615.4 1831.45
    3667 1832.18  3706.6 1831.22  3757.2 1831.63  3807.9  1830.1    4203 1829.19
  4288.4 1827.61  4416.7 1827.45  4456.3 1826.28    4588 1825.66  4601.6 1824.77
    4669 1825.39  4709.5    1824  4914.8  1822.5  5035.8 1822.95  5216.5  1821.9
  5216.8  1821.4  5220.5  1821.9  5414.4 1822.84  5572.9 1825.69  5703.7 1826.57
  5887.8 1826.88  5972.9 1828.88  6061.7 1828.36  6220.2 1831.17  6329.3  1831.3
#Mann= 5 ,-1 , 0
    3222    .045       0    3232     .07       0  5216.5     .07       0
  5220.5     .07       0  5703.7    .045       0
Bank Sta=5216.5,5220.5
XS Rating Curve= 0 ,0
Exp/Cntr=0.3,0.1

Type RM Length L Ch R = 1 ,38328   ,878,878,878
BEGIN DESCRIPTION:
Mapping XS 4abe1742
END DESCRIPTION:
XS GIS Cut Line= 3
      1510363.61      6856638.43      1511863.58      6856133.23
      1512721.49      6856008.45
#Sta/Elev= 30
  3385.7 1832.09  3545.4 1831.04  3851.5 1827.38  3875.2 1826.05  3969.7 1825.82
  4288.7 1822.27  4347.6 1822.34  4421.3 1820.08    4474 1819.86  4505.7 1820.69
  4523.3 1819.89    4589 1817.41  4695.6 1816.03  4737.7 1816.27  4769.5 1817.02
  4783.3 1815.86  4820.2 1815.31  4820.5 1814.81  4824.2 1815.31  4873.3 1817.41
  4917.2  1818.4  4935.4 1818.22  4940.7 1816.82  5010.3 1816.11  5081.1 1816.61
  5151.8 1815.33    5318 1816.96  5434.7 1817.02  5528.3 1818.79  5835.4 1818.77
#Mann= 7 ,-1 , 0
  3385.7    .125       0  4288.7    .094       0  4523.3    .035       0
  4737.7    .094       0  4820.2    .035       0  4824.2    .094       0
  4873.3    .035       0
Bank Sta=4820.2,4824.2
XS Rating Curve= 0 ,0
Exp/Cntr=0.3,0.1

Type RM Length L Ch R = 1 ,37450   ,676,676,676
BEGIN DESCRIPTION:
Mapping XS aa453712
END DESCRIPTION:
XS GIS Cut Line= 3
      1511233.81      6857142.78      1512202.56      6856736.53
      1512780.32      6856065.07
#Sta/Elev= 30
  3913.6 1822.53  4064.7 1820.61  4300.4 1819.22  4413.7 1817.43  4518.3 1816.71
  4543.8 1816.81  4636.5 1814.93  4852.5 1813.56  4866.5 1813.44  5007.2 1812.42
  5078.6 1813.18  5085.1 1812.19  5107.1 1813.12  5113.7 1812.49  5125.9 1809.27
  5126.2 1808.77  5129.7 1808.77  5129.9 1809.27  5134.5 1812.09  5142.2  1813.8
  5148.8 1813.13  5178.6 1813.07  5439.6 1813.62  5503.2 1814.88  5560.3    1815
    5603  1816.6  5666.7 1816.71  5743.3 1818.68  5815.9 1819.35  5849.9 1818.93
#Mann= 8 ,-1 , 0
  3913.6    .045       0  4518.3     .07       0  4852.5    .045       0
  4866.5     .07       0  5125.9     .07       0  5129.9     .07       0
  5178.6    .045       0  5743.3    .035       0
Bank Sta=5125.9,5129.9
XS Rating Curve= 0 ,0
Exp/Cntr=0.3,0.1

Type RM Length L Ch R = 1 ,36774   ,228,228,228
BEGIN DESCRIPTION:
Mapping XS 0a3dd68f
END DESCRIPTION:
XS GIS Cut Line= 3
      1512087.42      6857759.05      1512733.25      6857050.71
      1512927.69      6855988.22
#Sta/Elev= 30
  4011.8 1815.57    4230 1814.94  4294.1 1813.82    4386 1813.61  4520.5 1811.94
  4846.1 1809.74  4910.3  1810.5  4952.2 1811.03  4983.3 1808.85  4993.4 1806.42
  5001.2 1806.12  5001.4 1805.62  5005.2 1806.12  5008.3 1808.98  5013.8 1810.95
  5034.1 1810.09  5044.3 1811.07  5054.4 1810.59  5061.5  1808.6  5066.6 1808.59
  5084.9 1810.38  5135.8 1811.11  5347.9 1811.73  5572.9 1811.98  5644.1 1813.91
  5684.7 1813.56  5730.3  1814.3  5836.6 1816.94  5928.4 1817.03  6050.5 1816.61
#Mann= 6 ,-1 , 0
  4011.8    .045       0  4910.3     .07       0  5001.2     .07       0
  5005.2     .07       0  5347.9    .045       0  5928.4    .035       0
Bank Sta=5001.2,5005.2
XS Rating Curve= 0 ,0
Exp/Cntr=0.3,0.1

Type RM Length L Ch R = 1 ,36546   ,1018,1018,1018
BEGIN DESCRIPTION:
Mapping XS c909c914
END DESCRIPTION:
XS GIS Cut Line= 3
      1512622.15      6857988.18      1512886.03      6857224.33
      1513316.59      6855904.85
#Sta/Elev= 30
    4148 1810.72    4324 1810.87  4652.3 1808.73  4730.1 1808.84  4740.7 1807.65
  4749.9 1807.42  4761.8 1808.49  4781.1 1808.83  4825.3 1808.02  4843.5 1808.35
    4857 1807.64  4920.5 1806.82  4956.2 1807.32  4971.8 1804.53    4972 1804.03
  4975.5 1804.03  4975.8 1804.53  4994.4 1805.01  5000.4 1805.96  5037.6 1806.46
  5080.3 1808.54  5133.3 1807.28  5159.9  1808.3  5215.3 1808.81  5712.6 1809.84
  5776.4 1810.35  5814.8 1811.74  5888.5 1810.91    6206 1811.69  6344.1 1811.54
#Mann= 6 ,-1 , 0
    4148    .045       0  4652.3     .07       0  4971.8     .07       0
  4975.8     .07       0  5080.3    .045       0    6206    .035       0
Bank Sta=4971.8,4975.8
XS Rating Curve= 0 ,0
Exp/Cntr=0.3,0.1

Type RM Length L Ch R = 1 ,35528   ,987,987,987
BEGIN DESCRIPTION:
Mapping XS e8e2f806
END DESCRIPTION:
XS GIS Cut Line= 3
      1512685.05      6857974.54       1513775.2      6857487.51
      1514726.69      6855714.14
#Sta/Elev= 30
    3806 1810.35  4559.3 1805.28  4695.5 1804.99    4726 1803.46  4780.7 1804.54
  4886.6 1803.59  4909.8 1801.46    4933 1802.79    4945 1801.71  4984.9 1802.09
  4995.2 1800.69  4995.4 1800.19  4999.2 1800.69  5108.6 1803.08  5281.3  1802.8
  5347.1  1803.7  5390.9 1802.64  5749.2 1802.25  5963.4 1802.29  6343.5 1804.37
    6418 1805.19  6447.4 1806.81  6535.1 1806.45  6633.4    1809    6661  1808.3
  6758.5 1809.79  6786.8 1811.28  6918.1 1812.14  6972.8 1813.96  7012.5 1813.51
#Mann= 8 ,-1 , 0
    3806    .045       0  4559.3     .07       0  4995.2     .07       0
  4999.2     .07       0  5108.6    .045       0  5749.2     .07       0
  5963.4    .045       0  6918.1    .035       0
#XS Ineff= 2 , 0
       0                  5339.9       0    1805
Permanent Ineff=
       F       F
Bank Sta=4995.2,4999.2
XS Rating Curve= 0 ,0
Exp/Cntr=0.3,0.1

Type RM Length L Ch R = 1 ,34541   ,712,712,712
BEGIN DESCRIPTION:
Mapping XS 081eda1f
END DESCRIPTION:
XS GIS Cut Line= 4
       1512711.1      6858037.06      1514283.98      6858167.26
      1514638.15      6857859.97      1514888.14      6855734.98
#Sta/Elev= 30
  2930.8 1809.84  4229.1 1800.63  4269.3 1801.27  4601.8 1798.73  4771.4 1799.02
  4927.5  1799.1    4956 1799.59  4962.6 1801.08  4981.5 1800.69  4994.4 1799.22
  4998.1 1797.37  4998.3 1796.87  5002.1 1797.37  5040.3 1798.97  5684.8 1798.32
  5996.9 1798.84  6197.4 1800.45  6268.8 1801.95  6295.7 1801.44    6394 1802.87
  6520.5 1804.28  6580.9 1806.58    6601 1805.95  6691.7 1807.02  6752.1 1809.05
  6836.5  1809.4  6963.4 1811.43    7034 1813.97  7089.4 1813.45  7117.6 1814.26
#Mann= 10 ,-1 , 0
  2930.8    .045       0  4771.4     .07       0  4998.1     .07       0
  5002.1     .07       0  6197.4    .045       0  6295.7     .07       0
    6394    .045       0  6836.5     .07       0  6963.4    .045       0
  7089.4    .035       0
#XS Ineff= 2 , 0
       0  4962.6 1801.08               0
Permanent Ineff=
       F       F
Bank Sta=4998.1,5002.1
XS Rating Curve= 0 ,0
Exp/Cntr=0.3,0.1

Type RM Length L Ch R = 1 ,33829   ,713,713,713
BEGIN DESCRIPTION:
Mapping XS f76536da
END DESCRIPTION:
XS GIS Cut Line= 6
      1513072.74      6858123.53      1514286.28      6858180.82
      1514853.99      6857842.28      1515208.55      6857929.99
      1515281.07      6857659.98      1516228.32      6856702.33
#Sta/Elev= 30
    2482 1807.29  3786.5 1798.54    4228    1799  4243.9 1799.86  4275.1 1798.98
  4280.9 1796.98  4289.2 1796.51  4379.5 1797.36  4816.2 1795.68  4816.5 1795.18
  4820.6 1795.68  5105.9 1796.07  5298.2 1798.87    5410  1800.2  5431.1 1801.79
  5480.7 1801.64  5530.1 1804.01  5596.8 1804.28  5636.3 1806.03  5692.8 1805.96
  5735.3 1808.12  5756.4 1807.34  5855.4 1810.33  5890.8 1809.81  5955.8 1811.38
  5975.7 1812.57  6032.3 1812.43  6074.6 1814.46  6130.9 1814.63  6349.7 1820.58
#Mann= 8 ,-1 , 0
    2482    .045       0    4228     .07       0  4816.2     .07       0
  4820.6     .07       0  5298.2    .045       0  5596.8     .07       0
  5955.8    .045       0  6130.9     .07       0
Bank Sta=4816.2,4820.6
XS Rating Curve= 0 ,0
Exp/Cntr=0.3,0.1

Type RM Length L Ch R = 1 ,33116   ,168,168,168
BEGIN DESCRIPTION:
Mapping XS 8c20e4bb
END DESCRIPTION:
XS GIS Cut Line= 6
      1513153.32      6858149.03      1514286.15      6858196.78
      1514885.11      6857866.91      1515787.88      6858096.95
      1516781.81      6858300.94      1517231.62      6858158.21
#Sta/Elev= 30
  2245.3  1806.6  3291.2 1799.28  3472.4 1798.48  3678.8 1798.85  3841.6 1797.88
  3921.5 1798.27  3966.6 1798.86  3972.3 1799.89  3982.6 1799.98  4010.1 1797.43
  4026.2 1797.03  4573.6 1795.94  4609.3 1795.31    5026 1795.05  5193.5 1793.43
  5193.8 1792.93    5198 1793.43  5222.4 1794.48  5227.5 1793.78  5272.8 1794.92
    5424 1794.79  5614.3 1797.02  5634.7 1794.81    5676 1794.33  5736.8 1796.26
  5816.9 1797.02  5828.7 1796.13  5859.3 1797.25  6031.9 1798.51  6481.1 1809.11
#Mann= 4 ,-1 , 0
  2245.3    .045       0  3921.5     .07       0  5193.5     .07       0
    5198     .07       0
#XS Ineff= 2 , 0
       0                  5614.3       0 1797.02
Permanent Ineff=
       F       F
Bank Sta=5193.5,5198
XS Rating Curve= 0 ,0
Exp/Cntr=0.3,0.1

Type RM Length L Ch R = 1 ,32948   ,267,267,267
BEGIN DESCRIPTION:
Mapping XS b9f4343b
END DESCRIPTION:
XS GIS Cut Line= 4
      1513393.33      6858240.18      1515773.56      6858234.97
      1516841.27      6858427.68      1517179.84      6858266.21
#Sta/Elev= 30
  2587.9 1804.64  3169.6 1800.94  3219.6 1801.29  3399.6 1799.18  3670.6 1798.35
  3779.6 1798.24  4039.6 1795.67  4309.6 1794.32  4629.6 1793.97  4679.6 1793.28
  4709.6 1794.22  4729.6 1793.41  4769.6 1793.19  4949.6 1794.28  5091.5 1793.21
  5223.6 1793.67  5254.1 1793.15  5297.4  1793.2  5315.1 1794.57  5376.1 1793.21
  5404.5 1793.78  5426.9 1792.99  5578.1  1792.2  5578.4  1791.7  5582.3  1791.7
  5582.6  1792.2  5767.6 1794.92  5810.8 1795.39  6079.4 1798.63  6428.2 1807.34
#Mann= 6 ,-1 , 0
  2587.9    .045       0  3670.6     .07       0  5578.1     .07       0
  5582.6     .07       0  5767.6    .045       0  5810.8     .07       0
Bank Sta=5578.1,5582.6
XS Rating Curve= 0 ,0
Exp/Cntr=0.3,0.1

Type RM Length L Ch R = 1 ,32681   ,928,928,928
BEGIN DESCRIPTION:
Mapping XS 0e4bf138
END DESCRIPTION:
XS GIS Cut Line= 4
      1513914.06      6859486.21       1515897.6      6858461.88
      1516917.56      6858513.97      1517360.14      6858314.38
#Sta/Elev= 30
    2735 1804.35  2935.6 1801.55  3024.2    1802  3090.6 1800.17  3195.8 1800.64
  3544.6 1798.16  3602.7  1796.8  3699.6  1797.4  3921.1 1795.07  4054.1  1795.6
  4181.3 1793.43    4220 1794.52    4425 1791.75  4509.2 1792.15  4640.9 1792.03
  4694.4 1790.67  4812.5 1791.43  5265.2 1790.04  5345.3 1791.01  5373.1 1789.32
  5373.4 1788.82  5377.6 1789.32  5384.4 1790.27  5505.5 1793.32  5755.8 1795.24
  6021.2 1799.99  6128.5 1801.43    6141 1802.86  6210.4 1803.58  6474.2 1810.39
#Mann= 6 ,-1 , 0
    2735    .045       0  4509.2     .07       0  5373.1     .07       0
  5377.6     .07       0  5384.4    .045       0  6021.2     .07       0
Bank Sta=5373.1,5377.6
XS Rating Curve= 0 ,0
Exp/Cntr=0.3,0.1

Type RM Length L Ch R = 1 ,31753   ,680,680,680
BEGIN DESCRIPTION:
Mapping XS 34cb75ae
END DESCRIPTION:
XS GIS Cut Line= 3
      1514112.51      6859772.31      1516321.74      6858938.96
      1517431.38      6858375.47
#Sta/Elev= 30
  2649.7 1804.85    2802 1804.01  2848.1 1802.51  2933.3 1802.85  3013.2 1800.69
  3058.5 1801.36    3144  1799.6  3244.1 1799.96  3299.2 1798.52  3560.8 1797.24
  3835.6 1794.04  3934.9 1794.59  4041.8 1792.68  4105.9 1793.42    4170 1792.22
  4255.5 1792.75  4322.2 1791.35  4691.6 1789.89  4803.5 1788.29  4833.7 1789.54
  4883.4 1788.52  4885.3 1787.11  4885.8 1786.61  4892.3 1787.11  4907.5  1788.3
  4960.9 1787.19  5103.7 1789.12  5339.8 1791.66  5958.8 1803.09  6255.4 1811.06
#Mann= 6 ,-1 , 0
  2649.7    .045       0  4691.6     .07       0  4885.3     .07       0
  4892.3     .07       0  5103.7    .045       0  5958.8     .07       0
Bank Sta=4885.3,4892.3
XS Rating Curve= 0 ,0
Exp/Cntr=0.3,0.1

Type RM Length L Ch R = 1 ,31073   ,986,986,986
BEGIN DESCRIPTION:
Mapping XS 1502291e
END DESCRIPTION:
XS GIS Cut Line= 3
      1514286.71      6860179.13      1516296.28      6859480.34
      1517594.05      6858785.88
#Sta/Elev= 30
  2863.5 1804.95  2942.1 1805.68  3004.3 1803.88    3222 1802.28    3264  1800.6
  3335.8 1801.23  3380.5 1799.61  3921.5 1794.39  4040.7 1794.72  4584.7 1790.54
    4678 1790.43  4709.1 1792.53  4725.1 1790.43  4746.2 1789.81  4859.3 1789.24
  4946.8 1786.32  4968.6  1787.3  4987.8 1784.87  5022.9 1786.01  5024.9 1784.02
  5025.4 1783.52  5032.2 1784.02  5044.9 1786.08  5066.8 1786.71  5072.5 1785.11
  5088.7 1786.97  5183.4 1786.56  5443.3 1786.55  5613.4 1788.89    6463 1810.03
#Mann= 5 ,-1 , 0
  2863.5    .045       0  4946.8     .07       0  5024.9     .07       0
  5032.2     .07       0  5183.4    .045       0
Bank Sta=5024.9,5032.2
XS Rating Curve= 0 ,0
Exp/Cntr=0.3,0.1

Type RM Length L Ch R = 1 ,30087   ,781,781,781
BEGIN DESCRIPTION:
Mapping XS c38dce46
END DESCRIPTION:
XS GIS Cut Line= 3
       1515152.2      6860480.34      1516549.75      6860124.44
      1517747.62      6859377.93
#Sta/Elev= 30
    3552 1798.52  3622.1 1798.73    3689 1796.91  3944.1 1795.84    3985 1794.71
  4101.8 1794.72  4194.7 1792.95  4277.2 1794.02  4328.8 1792.08  4524.9    1791
  4925.4 1785.39  4956.3 1785.79  4968.6 1783.12  5001.6 1783.39  5007.3 1782.43
  5007.8 1781.93  5014.7 1782.43  5038.1 1784.04  5184.5 1783.96    5221 1782.59
  5242.3 1784.88  5278.9 1783.07  5315.4 1783.18  5321.3 1784.25    5437 1782.81
  5452.3 1783.42  5467.7 1786.17    5537 1786.57  6113.1 1796.47  6405.6 1803.12
#Mann= 5 ,-1 , 0
    3552    .045       0  4925.4     .07       0  5007.3     .07       0
  5014.7     .07       0    5537    .045       0
Bank Sta=5007.3,5014.7
XS Rating Curve= 0 ,0
Exp/Cntr=0.3,0.1

Type RM Length L Ch R = 1 ,29306   ,1814,1814,1814
BEGIN DESCRIPTION:
Mapping XS 39e47b5d
END DESCRIPTION:
XS GIS Cut Line= 4
      1515568.89      6861083.63      1516558.43       6860810.2
      1516909.99      6860549.78      1517764.12      6859491.88
#Sta/Elev= 30
  3542.6 1795.97  3623.4 1795.75  3657.7 1796.65  3683.8 1795.19  3797.9 1793.81
    3924 1793.61    4244 1790.69  4358.2 1790.76  4812.1 1784.48  4847.5 1785.02
  4868.4 1783.19  4894.5 1782.98  4927.4 1781.53  4997.8 1781.85  5014.2 1779.89
  5015.4 1779.84  5015.9 1779.34  5022.8 1779.84  5025.5 1780.86  5047.6 1782.44
  5103.8 1783.56    5211 1782.49  5479.1 1785.39  5879.4 1792.06  5957.8 1794.43
    5993 1794.38  6050.1 1796.32  6120.9 1796.86  6184.9 1798.98  6366.4 1802.13
#Mann= 7 ,-1 , 0
  3542.6    .045       0  4894.5     .07       0  4927.4    .045       0
  5014.2     .07       0  5015.4    .045       0  5022.8     .07       0
  5479.1    .045       0
Bank Sta=5015.4,5022.8
XS Rating Curve= 0 ,0
Exp/Cntr=0.3,0.1

Type RM Length L Ch R = 1 ,27492   ,423,423,423
BEGIN DESCRIPTION:
Mapping XS 6af4666c
END DESCRIPTION:
XS GIS Cut Line= 4
      1515729.48      6861265.93      1517313.64      6861109.68
      1517886.55      6860866.62      1518237.48      6859831.16
#Sta/Elev= 30
  3416.8 1795.11  3481.4 1793.75  3603.2 1792.39  3750.6  1792.2    4186 1789.12
  4336.8 1788.85  4507.6 1787.52    4799  1782.8  4881.8 1783.26  4939.7 1780.76
  4969.8 1777.99    4996 1777.69  4996.5 1777.19  5003.9 1777.69  5042.7  1778.8
  5086.2 1778.92  5102.5 1780.57  5155.3 1780.98  5202.6 1779.57    5208 1780.17
  5325.7 1781.19    5675 1783.51  6009.6 1788.36  6109.5 1788.83  6198.5 1791.55
    6298 1792.38  6549.3 1796.53  6575.5 1797.53  6612.1 1797.35  6724.3 1798.92
#Mann= 6 ,-1 , 0
  3416.8     .07       0  3481.4    .045       0  4881.8     .07       0
    4996     .07       0  5003.9     .07       0  5325.7    .045       0
Bank Sta=4996,5003.9
XS Rating Curve= 0 ,0
Exp/Cntr=0.3,0.1

Type RM Length L Ch R = 1 ,27069   ,499,499,499
BEGIN DESCRIPTION:
Mapping XS 2404acff
END DESCRIPTION:
XS GIS Cut Line= 4
      1516098.33       6861391.8      1517508.95       6861435.2
      1517953.28      6860883.93      1518302.23       6859915.2
#Sta/Elev= 30
  3592.5 1792.96  3627.9 1791.57  3632.9 1792.64  3639.2 1792.53  3709.2 1790.19
  3789.3  1791.6  3815.8 1790.88  3929.3 1789.46  4445.7 1787.42  4629.7 1786.07
  4706.5 1784.43  4828.5 1782.18  4879.8 1780.02  4919.8 1779.48  4949.8 1777.68
  4969.8 1778.37  4995.4 1776.92  4995.9 1776.42  5003.3 1776.92  5026.9 1778.79
  5084.4 1778.41  5148.4 1780.58    5235 1780.23  5404.3 1781.58  5546.7 1781.55
    5750 1783.43  6499.1  1792.8  6524.5 1794.09  6632.2 1795.67  6741.5 1796.03
#Mann= 8 ,-1 , 0
  3592.5     .07       0  3815.8    .045       0  4445.7     .07       0
  4706.5    .035       0  4828.5     .07       0  4995.4     .07       0
  5003.3     .07       0    5235    .045       0
Bank Sta=4995.4,5003.3
XS Rating Curve= 0 ,0
Exp/Cntr=0.3,0.1

Type RM Length L Ch R = 1 ,26570   ,1279,1279,1279
BEGIN DESCRIPTION:
Mapping XS befd9a34
END DESCRIPTION:
XS GIS Cut Line= 4
      1516997.65      6861892.67      1517836.21      6861882.25
      1518177.24      6860514.14      1518797.05      6860165.17
#Sta/Elev= 30
  3901.4 1786.87  4160.3 1786.87  4354.9 1785.75  4661.6  1782.4  4775.3 1781.67
  4799.1 1784.22  4835.2 1781.37  4922.9 1779.23  4996.4 1775.98  4996.9 1775.48
  5004.3 1775.98  5014.5 1777.94    5033  1779.1  5200.7 1779.11  5300.9 1779.48
  5401.2  1780.2  5461.4  1780.1  5501.4 1780.09  5859.7 1784.06    5871 1783.93
  6024.5 1786.01  6096.5 1787.19  6336.3 1787.25  6352.2 1785.79  6411.4 1784.33
  6439.4 1785.88  6498.1 1789.77    6555 1791.65  6631.3 1793.56  6861.3 1800.05
#Mann= 19 ,-1 , 0
  3901.4     .07       0  4160.3    .035       0  4354.9     .07       0
  4661.6    .035       0  4996.4    .035       0  5004.3    .035       0
  5014.5     .07       0  5200.7    .035       0  5300.9     .07       0
  5401.2    .045       0  5461.4     .07       0  5501.4    .045       0
  5859.7    .035       0    5871    .045       0  6024.5    .035       0
  6096.5    .045       0  6439.4    .035       0    6555    .045       0
  6631.3     .07       0
Bank Sta=4996.4,5004.3
XS Rating Curve= 0 ,0
Exp/Cntr=0.3,0.1

Type RM Length L Ch R = 1 ,25291   ,258,258,258
BEGIN DESCRIPTION:
Mapping XS 09552609
END DESCRIPTION:
XS GIS Cut Line= 4
      1517159.86      6861966.74      1518281.41       6861984.1
      1518763.29      6861215.58      1518935.17        6860377.
#Sta/Elev= 30
  2954.5 1786.85  3008.9 1786.93  3329.7 1785.72  3395.4 1784.61  3539.7 1783.94
  3649.7 1782.31  3879.8 1782.53  3991.4 1781.61  4083.4  1781.9    4112 1780.97
  4142.4 1782.54  4169.8 1780.79  4213.2 1781.78  4379.5 1780.93  4595.8 1778.38
  4863.9  1776.5    4924 1775.71  5011.4 1776.92  5017.6 1775.61  5018.1 1775.11
  5025.8 1775.61  5035.9 1776.02  5135.2 1777.61  5154.3 1778.94  5167.9 1782.96
  5263.6  1787.4  5566.1  1796.5  5731.6 1800.49  5777.2 1801.81  5839.3 1802.64
#Mann= 12 ,-1 , 0
  2954.5     .07       0  3008.9    .035       0  3395.4     .07       0
  3991.4    .035       0  4595.8     .07       0  4863.9    .035       0
  5017.6    .035       0  5025.8    .035       0  5035.9     .07       0
  5135.2    .035       0  5731.6     .07       0  5777.2    .035       0
Bank Sta=5017.6,5025.8
XS Rating Curve= 0 ,0
Exp/Cntr=0.3,0.1

Type RM Length L Ch R = 1 ,25033   ,849,849,849
BEGIN DESCRIPTION:
Mapping XS 1ab05a0e
END DESCRIPTION:
XS GIS Cut Line= 3
      1518630.01      6862362.97       1518912.6      6861420.44
      1519210.28      6860074.24
#Sta/Elev= 30
  3995.2 1780.08    4204 1778.98  4313.7 1777.04  4341.5  1779.1  4379.8 1776.89
  4605.9 1776.02    4679 1774.55  4863.7 1775.96  4883.7 1774.24  4884.2 1773.74
  4891.9 1774.24  4919.1 1775.49    4983  1774.3  5015.5 1776.89  5043.1 1775.71
  5135.3 1777.05    5207 1779.02  5236.3 1781.48  5292.7 1782.99  5360.6 1787.94
  5411.2 1789.36  5452.8 1790.54  5483.5 1794.75  5545.3  1796.1  5619.6 1797.44
  5798.4  1802.6  5803.5 1803.89  5821.5  1803.4  6199.6  1812.7  6357.9 1815.28
#Mann= 8 ,-1 , 0
  3995.2    .035       0  4883.7    .035       0  4891.9    .035       0
  5236.3     .07       0  5411.2    .035       0  5545.3     .07       0
  5619.6    .035       0  6199.6     .07       0
Bank Sta=4883.7,4891.9
XS Rating Curve= 0 ,0
Exp/Cntr=0.3,0.1

Type RM Length L Ch R = 1 ,24184   ,446,446,446
BEGIN DESCRIPTION:
Mapping XS 0a7dc2b2
END DESCRIPTION:
XS GIS Cut Line= 4
      1518680.01      6862412.96      1518804.33      6861999.98
      1519778.05      6862133.12      1520187.75      6861334.54
#Sta/Elev= 30
  4113.8 1778.53  4338.3 1778.13  4393.5 1777.06  4442.7 1777.53    4474 1776.51
  4492.5 1778.17  4530.8 1776.19  4547.9 1777.03    4722  1775.5  4785.9  1773.7
  4790.9 1774.47  4858.1    1773  4949.5 1772.44  4965.5 1770.97    4966 1770.47
  4973.9 1770.97  4989.9 1772.81  5017.9 1772.97  5322.9 1773.57  5383.9 1774.85
  5464.2 1774.19  5535.7 1774.76  5552.3    1776  5568.6 1775.52  5915.7 1781.97
  6084.9  1786.6  6206.8 1788.18  6264.2  1790.4  6417.6 1792.83  6425.4 1792.85
#Mann= 7 ,-1 , 0
  4113.8    .035       0    4722     .07       0  4965.5    .035       0
  4973.9     .07       0  5017.9     .07       0  5568.6    .045       0
  6417.6     .07       0
Bank Sta=4965.5,4973.9
XS Rating Curve= 0 ,0
Exp/Cntr=0.3,0.1

Type RM Length L Ch R = 1 ,23738   ,615,615,615
BEGIN DESCRIPTION:
Mapping XS 9742615b
END DESCRIPTION:
XS GIS Cut Line= 4
      1518780.01      6862412.99      1518965.55      6862251.17
      1519903.05      6862383.12      1520410.01      6861334.46
#Sta/Elev= 30
  4162.6 1777.74  4172.4 1777.72  4264.7  1777.4  4280.8 1777.73  4610.2 1775.81
  4882.9 1771.06  4997.5 1771.29  5014.2 1771.01  5030.1  1768.9  5030.6  1768.4
  5038.6  1768.9  5054.5 1770.65  5094.9 1771.57  5370.3 1773.65  5405.6  1773.3
  5427.9 1775.19  5459.5 1773.27  5478.3  1775.5  5480.7 1775.65  5555.4 1775.95
  5877.3 1781.71  6260.9 1791.77  6272.6 1793.51  6293.3 1792.63  6408.1 1796.66
  6425.2 1796.13  6447.8 1799.36  6470.4 1797.93  6510.7 1800.82  6520.3 1800.95
#Mann= 11 ,-1 , 0
  4162.6    .035       0  4172.4     .07       0  4264.7    .035       0
  4280.8     .07       0  5030.1     .07       0  5038.6     .07       0
  5370.3    .035       0  5478.3     .07       0  5480.7    .045       0
  6293.3     .07       0  6510.7    .035       0
Bank Sta=5030.1,5038.6
XS Rating Curve= 0 ,0
Exp/Cntr=0.3,0.1

Type RM Length L Ch R = 1 ,23123   ,376,376,376
BEGIN DESCRIPTION:
Mapping XS 4f95987e
END DESCRIPTION:
XS GIS Cut Line= 3
      1518722.53       6863445.6      1519986.38      6862737.28
      1520528.04      6861355.35
#Sta/Elev= 30
  3508.6 1780.57  3969.1 1777.73  4023.4 1778.36  4088.5 1776.72  4382.6 1775.28
  4471.9 1772.96  4508.7 1774.17  4807.5 1771.34  4959.7 1771.81    4988 1768.02
  4988.5 1767.52  5000.9 1768.02  5024.3 1770.43  5085.5 1772.56  5298.1  1774.7
  5332.6 1773.61  5364.8 1775.22  5386.3 1773.58  5404.1 1776.54  5417.1  1776.4
    5644 1779.35  6089.9 1790.29  6149.9 1793.36  6174.4 1792.38  6228.6 1794.38
  6277.5 1797.56  6288.5 1800.04  6312.7 1798.16  6374.4 1802.11  6441.7 1802.97
#Mann= 7 ,-1 , 0
  3508.6    .045       0  3969.1     .07       0    4988     .07       0
  5000.9     .07       0  5298.1    .035       0  5417.1    .045       0
  6089.9     .07       0
Bank Sta=4988,5000.9
XS Rating Curve= 0 ,0
Exp/Cntr=0.3,0.1

Type RM Length L Ch R = 1 ,22747   ,938,938,938
BEGIN DESCRIPTION:
Mapping XS 1d2ef92a
END DESCRIPTION:
XS GIS Cut Line= 4
      1520083.15       6864156.2      1520166.94      6863591.45
      1520250.27      6862994.23      1520784.99       6861285.9
#Sta/Elev= 30
    3778  1779.6  3978.4 1779.34  4031.5 1777.63  4487.1 1775.04  4639.3 1774.46
  4720.7  1773.4    4938  1770.7  4972.6 1768.48  4973.1 1767.98  4986.1 1768.48
  5000.4  1770.7  5054.7 1769.57  5114.4 1771.67    5207 1770.32  5476.2 1773.11
  5513.8 1773.86  5534.8 1775.75  5566.2  1774.6  5593.3 1776.05  5649.4 1775.56
  5849.1 1779.28  6276.9 1790.11  6331.1 1791.22    6352 1793.03  6373.1 1792.41
  6622.1  1797.6  6654.5 1800.37  6671.2 1799.89    6687 1799.13    6742 1801.46
#Mann= 11 ,-1 , 0
    3778    .045       0  4487.1     .07       0  4639.3     .16       0
  4720.7     .07       0  4972.6     .07       0  4986.1     .07       0
    5207    .045       0  5476.2    .035       0  5593.3    .045       0
  6276.9     .07       0  6671.2    .045       0
Bank Sta=4972.6,4986.1
XS Rating Curve= 0 ,0
Exp/Cntr=0.3,0.1

Type RM Length L Ch R = 1 ,21809   ,1482,1482,1482
BEGIN DESCRIPTION:
Mapping XS 7a74f305
END DESCRIPTION:
XS GIS Cut Line= 3
      1520680.82      6864765.08      1520798.88      6863431.73
      1521500.14       6861675.1
#Sta/Elev= 30
  3584.8 1783.22  3688.1 1780.71  3792.7 1781.12  3933.2 1778.62  4093.9 1779.12
  4145.7 1776.67  4244.4 1777.29  4332.2 1774.92    4395 1775.37  4455.3 1773.22
  4529.7 1772.99  4579.5 1773.31  4710.3 1770.74    4992 1769.03  5000.9 1766.32
  5001.4 1765.82  5014.5 1766.32  5024.3 1768.67  5184.5 1769.78  5522.4 1769.91
  5584.2 1772.35    5638 1771.62  5749.3  1773.3  5791.8 1774.36  5821.5 1777.53
  5853.4 1775.42  5875.3 1777.36  5893.7 1776.27  6348.7 1784.06  6814.8  1788.3
#Mann= 9 ,-1 , 0
  3584.8    .045       0  4332.2     .07       0  4529.7    .045       0
  4579.5     .07       0  5000.9     .07       0  5014.5     .07       0
  5184.5    .045       0  5749.3    .035       0  5893.7    .045       0
Bank Sta=5000.9,5014.5
XS Rating Curve= 0 ,0
Exp/Cntr=0.3,0.1

Type RM Length L Ch R = 1 ,20327   ,235,235,235
BEGIN DESCRIPTION:
Mapping XS 912f74fd
END DESCRIPTION:
XS GIS Cut Line= 3
      1521139.16      6865153.95       1521521.1      6864022.01
      1521784.99      6861994.25
#Sta/Elev= 30
  3789.3 1784.52  4238.8 1779.27  4365.5 1779.09  4659.4 1773.93  4829.9 1767.84
  4944.9 1767.05  4967.1 1765.47  4998.1 1766.55  5008.2 1765.64  5011.2  1763.5
  5011.7    1763  5025.3  1763.5  5028.3 1766.82  5078.7 1768.82    5351 1767.38
  5391.4 1765.03  5421.6 1767.35  5512.4 1768.97  5557.6 1768.04    5908 1770.35
  5976.2 1769.56  6056.1 1771.92  6198.1 1773.21  6237.7 1775.34  6304.5 1775.42
  6339.3 1778.91  6409.9 1779.19  6448.7 1781.42  6836.8 1786.56  7028.8  1786.9
#Mann= 8 ,-1 , 0
  3789.3    .045       0  4659.4     .07       0  5011.2     .07       0
  5025.3     .07       0  5557.6    .045       0  6237.7    .035       0
  6304.5     .07       0  6448.7    .045       0
Bank Sta=5011.2,5025.3
XS Rating Curve= 0 ,0
Exp/Cntr=0.3,0.1

Type RM Length L Ch R = 1 ,20092   ,1236,1236,1236
BEGIN DESCRIPTION:
Mapping XS 07915123
END DESCRIPTION:
XS GIS Cut Line= 3
      1521403.06      6865181.69       1521708.6      6864133.12
      1522138.89      6862411.97
#Sta/Elev= 30
  3840.4 1784.38  4452.1 1779.61  4521.3 1780.23    4618 1777.22  4690.2 1774.78
  4729.6 1768.43  4781.7 1768.68  4875.4 1765.55  4935.5 1767.15  5059.2 1766.72
  5082.2 1764.67  5092.5 1764.83  5100.4 1767.31  5133.7 1767.37  5329.5 1766.02
    5374 1764.16  5374.5 1763.66  5388.1 1764.16  5401.7 1766.72  5579.1 1766.57
  6186.1 1772.13  6246.9 1773.41  6267.6 1772.29  6288.2 1773.95  6319.1 1772.34
    6350 1776.53  6395.7 1776.87  6566.5    1782  6593.2 1781.57  6706.7 1783.01
#Mann= 8 ,-1 , 0
  3840.4    .045       0  4452.1     .07       0    5374     .07       0
  5388.1     .07       0  5579.1    .045       0  6186.1    .035       0
  6395.7     .07       0  6593.2    .045       0
Bank Sta=5374,5388.1
XS Rating Curve= 0 ,0
Exp/Cntr=0.3,0.1

Type RM Length L Ch R = 1 ,18856   ,808,808,808
BEGIN DESCRIPTION:
Mapping XS e74e4b56
END DESCRIPTION:
XS GIS Cut Line= 3
      1522082.74      6865297.28      1522421.28      6863760.83
      1522348.36      6862547.32
#Sta/Elev= 30
  3403.5 1786.61  4030.4 1783.25    4130 1780.44  4170.8 1779.05  4229.7 1773.06
  4247.2 1770.39  4293.6 1769.04  4314.1 1772.58  4319.7 1771.06  4406.3 1768.34
  4672.3 1764.58  4787.6 1763.03    4949  1763.9  5001.4  1763.1  5002.5 1760.85
    5003 1760.35  5016.9 1760.85  5039.7 1765.22  5159.9 1763.66  5312.8 1765.82
  5576.2 1768.26    5699 1769.43  5801.1 1771.59  5812.3 1770.66  5851.2 1771.63
  5871.2 1770.31  5901.3 1774.54  5921.3 1775.64  6050.6 1780.13  6192.5 1781.85
#Mann= 13 ,-1 , 0
  3403.5    .045       0  4030.4     .07       0    4130    .035       0
  4229.7     .07       0  4247.2    .035       0  4672.3     .07       0
  5002.5     .07       0  5016.9     .07       0  5312.8    .045       0
  5576.2     .07       0    5699    .045       0  5812.3    .035       0
  6050.6     .07       0
Bank Sta=5002.5,5016.9
XS Rating Curve= 0 ,0
Exp/Cntr=0.3,0.1

Type RM Length L Ch R = 1 ,18048   ,1339,1339,1339
BEGIN DESCRIPTION:
Mapping XS 9e2bfa7d
END DESCRIPTION:
XS GIS Cut Line= 3
      1522348.36      6865364.99      1522988.34      6864071.34
      1522770.23      6862293.77
#Sta/Elev= 30
  3556.7 1786.09    3888 1784.76  4193.4 1780.15  4265.3 1777.02  4372.8 1774.72
    4409  1772.8  4459.1 1772.08  4738.9 1765.89  4916.8 1762.28  4939.2 1761.45
  4947.9 1759.85  4956.1 1762.16  4978.5 1761.73  4991.9 1758.69  4992.4 1758.19
  5006.3 1758.69  5033.6 1762.33  5068.7 1761.55  5086.4 1763.01  5231.4 1764.24
  5318.4 1762.38  5996.5 1767.74    6031 1767.23  6061.2 1769.31  6091.5 1767.51
  6115.6 1767.98  6403.8 1769.42  6705.8 1774.19  6736.3  1775.9  6790.9 1775.26
#Mann= 13 ,-1 , 0
  3556.7    .045       0  4193.4     .07       0  4265.3    .035       0
    4409     .07       0  4459.1    .035       0  4738.9     .07       0
  4947.9    .035       0  4991.9    .035       0  5006.3    .035       0
  5086.4     .07       0  5318.4    .045       0  5996.5    .035       0
  6115.6     .07       0
Bank Sta=4991.9,5006.3
XS Rating Curve= 0 ,0
Exp/Cntr=0.3,0.1

Type RM Length L Ch R = 1 ,16709   ,1084,1084,1084
BEGIN DESCRIPTION:
Mapping XS 79cefe73
END DESCRIPTION:
XS GIS Cut Line= 3
      1522942.81       6865500.4      1523802.18       6864345.9
      1523819.54      6862705.23
#Sta/Elev= 30
  3003.6 1782.16  3442.9 1782.72  3464.7 1783.91  3484.4 1782.77  3800.5 1779.52
  3921.4  1775.1  3942.3 1773.27  3956.9 1770.45  3992.3 1768.31  4039.3 1767.97
  4201.3 1765.01  4415.3 1761.82  4726.9 1761.31  4850.8 1760.83  4920.8 1762.05
  4980.8 1758.88  5000.8 1759.18  5003.2 1757.31  5003.7 1756.81  5018.3 1757.31
  5030.8 1760.67  5129.2 1761.37  5500.8 1765.56  5520.8  1764.8  5528.8  1765.9
  5570.8 1764.92  5590.8  1767.3  5626.7  1766.7  5970.8 1769.28  6083.6 1768.94
#Mann= 10 ,-1 , 0
  3003.6    .045       0  3484.4     .07       0  4039.3    .035       0
  4201.3    .045       0  4726.9     .07       0  5003.2     .07       0
  5018.3     .07       0  5129.2    .045       0  5528.8    .035       0
  5626.7    .045       0
Bank Sta=5003.2,5018.3
XS Rating Curve= 0 ,0
Exp/Cntr=0.3,0.1

Type RM Length L Ch R = 1 ,15625   ,918,918,918
BEGIN DESCRIPTION:
Mapping XS f5fc9dce
END DESCRIPTION:
XS GIS Cut Line= 3
      1523211.89      6865578.55      1524340.37      6864458.75
      1525416.76      6862314.65
#Sta/Elev= 30
  2934.6 1781.08  3128.1 1781.68  3361.5 1779.03  3389.8  1776.9  3764.5 1767.96
  4153.4 1761.99  4521.1 1759.43  4894.5 1759.23  4952.9 1757.63  4973.9 1756.04
  4990.6 1758.47  4996.2 1756.24  5012.9 1759.01  5027.7 1754.46  5028.2 1753.96
  5042.8 1754.46  5057.6 1757.87  5319.7 1758.21  5364.4 1756.92  5398.2 1759.39
    5521 1761.43  5554.6 1763.69  5568.5 1762.74  5609.9 1763.67  5660.6 1766.01
  5749.9 1764.72  6174.3 1768.53  6584.1 1772.86  6735.2 1776.07  6923.5 1780.57
#Mann= 7 ,-1 , 0
  2934.6    .045       0  4952.9     .07       0  5027.7     .07       0
  5042.8     .07       0  5568.5    .035       0  5609.9    .045       0
  6735.2     .07       0
Bank Sta=5027.7,5042.8
XS Rating Curve= 0 ,0
Exp/Cntr=0.3,0.1

Type RM Length L Ch R = 1 ,14707   ,130,130,130
BEGIN DESCRIPTION:
Mapping XS 79d956a1
END DESCRIPTION:
XS GIS Cut Line= 5
      1524943.61      6866119.29       1525275.2      6864466.71
      1525275.14      6864236.79      1525089.14      6863861.35
      1525512.26        6862549.
#Sta/Elev= 30
  3085.8 1761.75  3166.4 1760.25  3178.9 1761.41  3209.5 1760.09  3573.7 1757.41
    4114 1756.58  4382.6 1756.38  4786.7 1755.89    4920 1755.76  4962.4 1752.67
  4962.9 1752.17  4977.7 1752.67  5009.1 1755.18  5156.1 1755.49  5178.4  1757.8
    5426 1758.79  5465.8 1762.02  5484.9 1762.37  5497.3 1760.55  5507.8 1760.53
    5650 1765.41    5739 1766.35  5751.8 1765.37  5762.3  1766.8  5791.5 1766.04
  6064.7 1767.85  6136.5 1767.32  6474.4 1771.36  6654.3  1775.3  6799.1 1778.27
#Mann= 9 ,-1 , 0
  3085.8    .035       0    4114    .045       0  4382.6    .035       0
  4786.7     .07       0  4962.4     .07       0  4977.7     .07       0
    5650    .035       0  5762.3    .045       0  6654.3     .07       0
Bank Sta=4962.4,4977.7
XS Rating Curve= 0 ,0
Exp/Cntr=0.3,0.1

Type RM Length L Ch R = 1 ,14577   ,1941,1941,1941
BEGIN DESCRIPTION:
Mapping XS 938b5054
END DESCRIPTION:
XS GIS Cut Line= 4
      1525068.61      6866265.11      1525419.02      6864466.19
      1525394.72       6864077.3      1525656.61      6862571.49
#Sta/Elev= 30
  2943.2 1761.69    3032 1759.98  3772.7 1755.05    3784 1753.87  3788.4 1751.48
  3788.9 1750.98  3803.7 1751.48  3816.4 1755.26  3901.6 1756.92  4311.3 1754.83
  4465.5 1755.36    4522 1755.64  4580.5 1753.94  4723.1 1754.45  4743.5 1755.74
  4814.2 1754.99  4864.3  1756.6  4964.5 1754.32 4983.261752.085 4992.851752.257
  4994.5 1754.08  5004.6 1755.14  5064.7  1757.8  5551.1 1763.57  5605.7    1763
  5648.5 1764.67  5733.3 1764.33    6322 1769.79  6505.5 1774.06    6694 1779.56
#Mann= 9 ,-1 , 0
  2943.2    .045       0  3772.7     .07       0  3788.4    .035       0
  3803.7     .07       0  3901.6    .035       0  4311.3     .16       0
  4465.5    .035       0  5648.5    .045       0  6505.5     .07       0
#XS Ineff= 2 , 0
       0  3949.1 1757.62               0
Permanent Ineff=
       F       F
Bank Sta=4983.26,4992.85
XS Rating Curve= 0 ,0
Exp/Cntr=0.3,0.1

Type RM Length L Ch R = 1 ,12636   ,966,966,966
BEGIN DESCRIPTION:
Mapping XS 355ee160
END DESCRIPTION:
XS GIS Cut Line= 3
      1525328.14      6867123.87      1526114.77      6865437.96
      1526430.01      6863812.95
#Sta/Elev= 30
  3139.6 1786.05  3201.3 1776.04  3262.1 1772.41  3358.3 1768.92  3609.5 1762.23
  3764.2 1760.43  3827.3 1758.42  4006.8 1756.78  4106.1 1757.21  4329.4 1753.96
  4503.4 1753.42  4547.5 1751.53  4637.6 1750.46  4757.5 1751.99  4917.5 1750.02
  4963.2 1750.96  5009.1 1747.37  5018.1 1746.37  5018.6 1745.87  5034.7 1746.37
  5078.2  1746.9    5112 1749.17  5142.6 1754.82  5181.6 1752.14  5224.5 1752.51
  5760.7 1757.97  6526.4  1763.1  6551.8 1764.14  6622.4 1763.22  6655.3 1763.28
#Mann= 8 ,-1 , 0
  3139.6     .07       0  3358.3    .045       0  5009.1     .07       0
  5018.1    .045       0  5034.7     .07       0  5224.5    .045       0
  6526.4    .035       0  6622.4    .045       0
Bank Sta=5018.1,5034.7
XS Rating Curve= 0 ,0
Exp/Cntr=0.3,0.1

Type RM Length L Ch R = 1 ,11670   ,1107,1107,1107
BEGIN DESCRIPTION:
Mapping XS ca9d1357
END DESCRIPTION:
XS GIS Cut Line= 3
      1525598.97      6867540.52      1526925.38      6865769.67
      1527064.27      6864102.97
#Sta/Elev= 30
  2777.4 1772.06  2787.5 1771.65    2983 1768.77  3268.5 1762.48  3341.4 1762.23
  3397.7 1760.31  3476.8 1760.56  4933.3  1748.8  4968.8 1747.92  4977.2 1745.02
  4979.4 1743.81  4979.9 1743.31  4996.3 1743.81  5001.6  1746.1  5011.7 1746.47
  5081.9 1747.19    5122 1749.17  5161.6 1748.89  5172.2 1750.19  5182.3 1749.05
  5222.4 1749.21  5281.1 1751.89  5312.7 1749.69  5764.5 1755.21  5892.9 1756.02
  5903.5 1756.25  6045.1 1756.76  6143.2 1757.94  6282.5 1759.43  6662.4 1762.94
#Mann= 12 ,-1 , 0
  2777.4     .07       0  2787.5    .045       0  4977.2     .07       0
  4979.4     .07       0  4996.3     .07       0  5281.1    .045       0
  5764.5     .07       0  5892.9    .045       0  5903.5     .07       0
  6045.1    .045       0  6143.2     .07       0  6282.5    .045       0
Bank Sta=4979.4,4996.3
XS Rating Curve= 0 ,0
Exp/Cntr=0.3,0.1

Type RM Length L Ch R = 1 ,10563   ,1499,1499,1499
BEGIN DESCRIPTION:
Mapping XS ef6ac62e
END DESCRIPTION:
XS GIS Cut Line= 4
      1525844.86      6868413.46      1527418.21      6866319.28
      1527722.03      6865342.72        1527430.      6864363.01
#Sta/Elev= 30
  2366.2 1789.35  2612.4 1782.71  2748.3 1774.04  2812.3 1771.32  3091.4 1763.68
  3120.6 1764.15  3182.1 1761.56  3485.1 1758.15  3655.9 1758.28  3712.1 1756.64
    4112 1755.45  4749.4 1750.94  4862.1 1747.56  4988.6  1746.4  4988.8 1740.89
  4989.3 1740.39  5005.9 1740.89  5007.8 1743.78  5049.7 1745.72  5094.7 1746.56
  5162.8 1745.18  5615.3 1747.98  5782.8 1747.71  5950.4 1750.43  6329.3 1752.62
  6525.7 1754.52    6730 1755.83  6748.1 1755.88  6866.1  1756.5  7030.6 1758.74
#Mann= 10 ,-1 , 0
  2366.2     .07       0  3182.1    .045       0  4988.8     .07       0
  5005.9    .045       0  5162.8    .045       0  6329.3     .07       0
  6525.7    .045       0    6730     .07       0  6748.1    .045       0
  6866.1     .07       0
Bank Sta=4988.8,5005.9
XS Rating Curve= 0 ,0
Exp/Cntr=0.3,0.1

Type RM Length L Ch R = 1 ,9064    ,1803,1803,1803
BEGIN DESCRIPTION:
Mapping XS 34bc8ad6
END DESCRIPTION:
XS GIS Cut Line= 3
      1525975.08      6868597.92      1528180.39      6866508.35
      1528520.33       6865627.3
#Sta/Elev= 30
  1927.5 1787.33  1947.1 1787.23  2082.9    1785  2261.2 1775.31  2300.9 1774.71
  2330.5 1773.81  2351.9 1769.74  2409.3 1768.65  2607.7 1764.16  2794.7 1760.72
    3222 1755.45  3724.1  1753.4  4015.9 1748.67  4466.8 1742.79  4586.9 1743.14
  4615.2 1747.03  4677.4 1736.55  4677.9 1736.05  4694.6 1736.55  4735.8 1743.67
  4778.2 1744.41  4841.7 1742.65  4961.9  1744.9  4976.6 1739.19  4987.1  1738.9
  4998.1 1742.36  5022.4 1743.25  5265.8 1744.11  5524.4 1748.72  5909.9 1750.94
#Mann= 11 ,-1 , 0
  1927.5    .045       0  1947.1     .07       0  2261.2    .035       0
  2300.9     .07       0  2409.3    .035       0  2607.7     .07       0
  2794.7    .045       0  4015.9     .07       0  4677.4     .07       0
  4694.6     .07       0  5265.8    .045       0
Bank Sta=4677.4,4694.6
XS Rating Curve= 0 ,0
Exp/Cntr=0.3,0.1

Type RM Length L Ch R = 1 ,7261    ,1159,1159,1159
BEGIN DESCRIPTION:
Mapping XS 04c5efec
END DESCRIPTION:
XS GIS Cut Line= 4
      1528286.26      6870192.98      1528173.45      6868195.85
      1528423.45       6867438.9      1528770.33      6865919.58
#Sta/Elev= 30
  2307.6 1764.92  2853.5 1762.28  3554.6 1752.67  3634.7 1753.31  3821.3 1749.79
  3895.1 1749.23  3905.1 1747.93  3934.3 1748.75  3945.2 1746.84  4065.4 1743.13
  4191.2  1741.1  4527.2  1740.4  4579.1 1741.46  4616.1 1739.97  4895.4 1740.45
  4948.1 1739.73  4965.2 1738.12  4979.7 1739.05  4980.4 1736.42  4980.9 1735.92
  4999.9 1736.42  5002.2 1738.56  5104.3 1743.37  5406.3 1745.01  5565.1 1744.27
  5717.4 1743.15  6028.5 1743.84  6418.9 1748.54  6511.3 1751.13  6663.5 1751.12
#Mann= 8 ,-1 , 0
  2307.6    .045       0  3821.3    .035       0  3934.3    .045       0
  4527.2     .07       0  4980.4     .07       0  4999.9     .07       0
  5104.3    .045       0  5565.1     .07       0
Bank Sta=4980.4,4999.9
XS Rating Curve= 0 ,0
Exp/Cntr=0.3,0.1

Type RM Length L Ch R = 1 ,6102    ,835,835,835
BEGIN DESCRIPTION:
Mapping XS f0dc67e0
END DESCRIPTION:
XS GIS Cut Line= 3
      1528361.42      6869594.17      1528921.32      6867710.46
      1528938.69      6867055.05
#Sta/Elev= 30
  3011.6 1760.24  3214.1 1758.46  3252.5 1756.69  3318.9 1756.87  3508.4 1752.82
  3600.2 1753.23  3737.9 1750.28  3848.4 1750.11  3862.5 1750.34  3886.6 1751.14
  3914.6 1748.88  4167.8 1745.32  4406.7 1738.14  4686.7 1740.32  4697.7 1738.24
  4749.8 1739.72  4822.8 1738.71  4835.1 1736.32  4843.7 1740.02    4875 1737.48
  4980.5 1739.13  4999.5  1734.7    5000  1734.2    5019  1734.7  5019.2 1737.65
  5029.2 1739.97  5069.3  1741.7  5319.3 1743.81  5514.9  1747.8  5632.4 1748.97
#Mann= 7 ,-1 , 0
  3011.6    .045       0  3848.4    .035       0  3862.5    .045       0
  4406.7     .07       0  4999.5     .07       0    5019     .07       0
  5514.9    .045       0
Bank Sta=4999.5,5019
XS Rating Curve= 0 ,0
Exp/Cntr=0.3,0.1

Type RM Length L Ch R = 1 ,5267    ,682,682,682
BEGIN DESCRIPTION:
Mapping XS 52b3c4c1
END DESCRIPTION:
XS GIS Cut Line= 3
      1528475.53      6870298.82      1529544.97      6868215.49
      1529230.01      6866913.02
#Sta/Elev= 30
  2311.1 1764.03    2638    1762  2696.5 1760.08  2779.6 1760.33  3008.9  1756.3
  3084.7 1756.47  3134.6 1754.56  3195.6 1754.97  3677.7 1748.83  3786.2 1748.52
  4234.2 1738.67  4604.3 1736.98  4907.5 1737.95    4968 1736.45  4989.8 1734.57
  5000.1 1731.72  5000.6 1731.22  5019.6 1731.72    5031 1736.68  5133.9 1737.07
  5145.7 1741.21  5154.4 1739.76  5164.7 1735.12  5195.6 1733.27  5224.2 1735.77
  5229.4 1737.87  5465.6 1742.28    5653 1745.53  5794.1 1745.62  5992.9 1747.62
#Mann= 8 ,-1 , 0
  2311.1    .045       0  3677.7    .035       0  3786.2    .045       0
  4604.3     .07       0  5000.1     .07       0  5019.6     .07       0
  5465.6    .045       0  5794.1     .07       0
#XS Ineff= 2 , 0
       0                  5145.7       0 1741.21
Permanent Ineff=
       F       F
Bank Sta=5000.1,5019.6
XS Rating Curve= 0 ,0
Exp/Cntr=0.3,0.1
