--- MULBERRY CREEK TRIBUTARY 21A.prj (project) ---

Proj Title=MULBERRY CREEK TRIBUTARY 21A Base Level Engineering
Current Plan=p01
Default Exp/Contr=0.3,0.1
English Units
Geom File=g01
Flow File=f01
Plan File=p01
Y Axis Title=Elevation
X Axis Title(PF)=Main Channel Distance
X Axis Title(XS)=Station
BEGIN DESCRIPTION:
MULBERRY CREEK TRIBUTARY 21A
END DESCRIPTION:
DSS File=dss
DSS Export Rating Curves= 0
DSS Export Rating Curve Sorted= 0
DSS Export Volume Flow Curves= 0
DXF OffsetX= 0
DXF OffsetY= 0
DXF ScaleX= 1
DXF ScaleY= 10

--- MULBERRY CREEK TRIBUTARY 21A.p01 (plan) ---

Plan Title=Multiple Run
Program Version=4.10
Short Identifier=Multiple Run
Geom File=g01
Flow File=f01
Subcritical Flow
K Sum by GR= 0
Std Step Tol= 0.01
Critical Tol= 0.01
Num of Std Step Trials= 20
Max Error Tol= 0.3
Flow Tol Ratio= 0.001
Split Flow NTrial= 30
Split Flow Tol= 0.02
Split Flow Ratio= 0.02
Log Output Level= 0
Friction Slope Method= 1
Unsteady Friction Slope Method= 2
Unsteady Bridges Friction Slope Method= 1
Parabolic Critical Depth
Global Vel Dist= 1 , 1 , 1
Global Log Level= 0
CheckData=True
Encroach Param=-1 ,0,0, 0
BEGIN DESCRIPTION:
Multiple Run
END DESCRIPTION:
Computation Interval=1HOUR
Output Interval=1HOUR
Run HTab= 0
Run UNet= 0
Run PostProcess= 0
Run WQNet= 0
UNET Theta= 1
UNET Theta Warmup= 1
UNET ZTol= 0.02
UNET ZSATol= 0.05
UNET MxIter= 20
UNET MaxInSteps= 0
UNET DtIC= 0
UNET DtMin= 0
UNET MaxCRTS= 20
UNET WFStab= 2
UNET SFStab= 1
UNET WFX= 1
UNET SFX= 1
UNET DSS MLevel= 4
UNET DZMax Abort= 100
UNET Convert EG Bridges= 0
UNET Use Existing IB Tables=-1
UNET Froude Reduction=False
UNET Froude Limit= 1
UNET Froude Power= 10
UNET Time Slicing=0,0, 5
UNET Junction Losses=0
Instantaneous Interval=1HOUR
DSS File=dss
Write IC File= 0
Write IC File at Sim End=0
Echo Input=False
Echo Parameters=False
Echo Output=False
Write Detailed= 0
WQ AD Non Conservative
WQ ULTIMATE=-1
WQ Max Comp Step=1HOUR
WQ Output Interval=15MIN
WQ Output Selected Increments= 0
WQ Output face flow=0
WQ Output face velocity=0
WQ Output face area=0
WQ Output face dispersion=0
WQ Output cell volume=0
WQ Output cell surface area=0
WQ Output cell continuity=0
WQ Output cumulative cell continuity=0
WQ Output face conc=0
WQ Output face dconc_dx=0
WQ Output face courant=0
WQ Output face peclet=0
WQ Output face adv mass=0
WQ Output face disp mass=0
WQ Output cell mass=0
WQ Output cell source sink temp=0
WQ Output cell source sink nsm=0
WQ Output MaxMinRange=-1
WQ Daily Max Min Mean=-1
WQ Daily Range=0
WQ Daily Time=0
WQ Create Restart=0
WQ Fixed Restart=0
WQ System Summary=0
WQ Use Fixed Temperature=0
Sorting and Armoring Iterations= 10
XS Update Threshold= 0.02
Hydraulics Update Threshold= 0.02
Energy Slope Method= 1
Volume Change Method= 0
XS Weighting Method= 0
Number of US Weighted Cross Sections= 1
Number of DS Weighted Cross Sections= 1
Upstream XS Weight=0.25
Main XS Weight=0.5
Downstream XS Weight=0.25
Number of DS XS's Weighted with US Boundary= 1
Upstream Boundary Weight= 1
Weight of XSs Associated with US Boundary= 0
Number of US XS's Weighted with DS Boundary= 1
Downstream Boundary Weight= 0.5
Weight of XSs Associated with DS Boundary= 0.5
Sediment Output Level= 4
Mass or Volume Output= 0
Output Increment Type= 1
Profile and TS Output Increment= 10
XS Output Flag= 0
XS Output Increment= 10
Disregard all LS=0
Disregard all Conn=0
Disregard all Breaches=0
Disregard all Pumps=0

--- MULBERRY CREEK TRIBUTARY 21A.f01 (steady flow) ---

Flow Title=Multiple
Program Version=4.10
Number of Profiles= 7
Profile Names=10-year,25-year,50-year,1pct_min,100-year,1pct_plu,500-year
River Rch & RM=MULBERRY CREEK T,Reach-1         ,30073
     315     454     573     361     720    1437    1150
River Rch & RM=MULBERRY CREEK T,Reach-1         ,28565
     538     798    1029     660    1317    2627    2183
River Rch & RM=MULBERRY CREEK T,Reach-1         ,25791
     681    1020    1321     851    1698    3388    2840
River Rch & RM=MULBERRY CREEK T,Reach-1         ,19768
    1078    1649    2168    1414    2822    5630    4843
River Rch & RM=MULBERRY CREEK T,Reach-1         ,16201
    1096    1672    2193    1427    2846    5679    4859
River Rch & RM=MULBERRY CREEK T,Reach-1         ,9089
    1138    1733    2269    1474    2941    5869    5005
River Rch & RM=MULBERRY CREEK T,Reach-1         ,1364
    1582    2443    3230    2117    4223    8426    7313
Boundary for River Rch & Prof#=MULBERRY CREEK T,Reach-1         , 1
Up Type= 0
Dn Type= 3
Dn Slope=0.00571
Boundary for River Rch & Prof#=MULBERRY CREEK T,Reach-1         , 2
Up Type= 0
Dn Type= 3
Dn Slope=0.00571
Boundary for River Rch & Prof#=MULBERRY CREEK T,Reach-1         , 3
Up Type= 0
Dn Type= 3
Dn Slope=0.00571
Boundary for River Rch & Prof#=MULBERRY CREEK T,Reach-1         , 4
Up Type= 0
Dn Type= 3
Dn Slope=0.00571
Boundary for River Rch & Prof#=MULBERRY CREEK T,Reach-1         , 5
Up Type= 0
Dn Type= 3
Dn Slope=0.00571
Boundary for River Rch & Prof#=MULBERRY CREEK T,Reach-1         , 6
Up Type= 0
Dn Type= 3
Dn Slope=0.00571
Boundary for River Rch & Prof#=MULBERRY CREEK T,Reach-1         , 7
Up Type= 0
Dn Type= 3
Dn Slope=0.00571
DSS Import GetInterval= 0
DSS Import GetPeak= 0
DSS Import FillOption= 0

--- MULBERRY CREEK TRIBUTARY 21A.g01 (geometry) ---

Geom Title=Existing Conditions
Program Version=4.10

River Reach=MULBERRY CREEK T,Reach-1
Reach XY= 30
        1462905.        6801188.      1462963.04      6802691.32
       1463445.9      6802831.29      1463306.96      6803182.11
       1463962.8      6804694.21      1465349.41      6805493.61
      1465460.83       6806340.3      1466191.44      6807024.51
      1467107.67      6807143.42      1467159.99        6807533.
      1467699.53      6807885.55      1467710.95      6810032.31
      1468211.34      6810045.36      1469552.57       6811382.6
      1470118.22      6811301.62      1470407.08      6812575.99
       1471121.2      6813754.71      1472368.35      6814351.36
      1472613.46       6815034.5      1473746.05      6815281.31
      1473607.06      6815832.15      1474151.25      6816489.55
      1474354.62      6817653.27      1474105.07      6818258.03
      1474253.95      6819027.56      1473831.88      6819811.83
      1473202.63      6819893.67      1473054.92      6820218.12
      1473404.99      6820480.47        1474055.        6820338.

Type RM Length L Ch R = 1 ,30073   ,686,686,686
BEGIN DESCRIPTION:
MULBERRY CREEK TRIBUTARY 21A 57.0
END DESCRIPTION:
XS GIS Cut Line= 3
      1462352.68      6801439.53      1462955.08      6801387.97
      1463680.43      6801166.21
#Sta/Elev= 30
  4395.4 2352.46  4447.9 2352.83  4467.5 2348.97  4478.5  2343.6  4518.2 2336.29
  4548.3 2320.74  4578.4 2310.66  4630.3 2306.78  4648.6  2303.6  4729.9 2300.33
  4849.4 2293.57  4909.6 2292.78  4959.8 2288.51  4983.4 2283.96  5008.4 2277.36
  5008.6 2276.86  5012.4 2277.36  5049.1 2288.61  5145.5 2290.84  5240.4 2297.09
  5282.3    2295    5351 2303.19  5397.9 2308.31  5418.2 2313.25  5470.5 2338.72
    5491 2343.42  5501.9 2348.74  5534.2 2354.23    5731 2361.03  5758.5 2367.22
#Mann= 9 ,-1 , 0
  4395.4     .16       0  4478.5     .07       0  4630.3     .16       0
  4729.9     .07       0  4983.4     .16       0  5008.4     .07       0
  5012.4     .16       0  5145.5    .035       0    5351     .16       0
Bank Sta=5008.4,5012.4
XS Rating Curve= 0 ,0
Exp/Cntr=0.3,0.1

Type RM Length L Ch R = 1 ,29387   ,539,539,539
BEGIN DESCRIPTION:
Mapping XS e056810e
END DESCRIPTION:
XS GIS Cut Line= 3
       1462226.8      6801756.38      1462968.99      6802029.81
      1463815.32      6801947.35
#Sta/Elev= 30
  4173.3 2340.31    4214 2338.18  4235.3 2334.21  4250.8 2330.32  4275.9    2321
  4320.6 2311.06  4438.4 2299.42  4827.8 2275.89  4964.3 2275.43  5018.5  2270.4
  5018.8  2269.9  5022.5  2270.4  5035.1  2270.6  5080.8 2276.68    5176 2278.97
  5287.8 2282.05  5382.2 2284.07  5412.4 2287.32  5452.6 2284.93  5472.7 2290.39
  5505.5 2294.93  5573.1  2307.7  5593.2 2313.13  5613.3  2320.3  5663.6 2344.49
  5683.7 2351.44  5733.9 2359.52  5757.7 2361.56  5774.1 2366.74  5814.6 2372.49
#Mann= 7 ,-1 , 0
  4173.3     .16       0  4438.4     .07       0  5018.5     .07       0
  5022.5     .07       0    5176     .16       0  5287.8    .035       0
  5505.5     .16       0
Bank Sta=5018.5,5022.5
XS Rating Curve= 0 ,0
Exp/Cntr=0.3,0.1

Type RM Length L Ch R = 1 ,28848   ,283,283,283
BEGIN DESCRIPTION:
Mapping XS 936d4803
END DESCRIPTION:
XS GIS Cut Line= 3
      1461863.13      6802257.25      1462713.78      6802472.52
      1463866.53      6802278.08
#Sta/Elev= 30
    3883 2353.36  3895.2 2352.86  3926.2 2343.22  3949.6 2340.84  3998.4 2323.39
  4024.2 2317.78    4050 2311.71  4091.2 2305.57  4236.7 2294.06  4758.5 2269.18
  4982.8 2263.62  4983.1 2263.12  4986.8 2263.62    5115 2267.49  5368.9 2268.78
  5461.5 2271.21  5546.3 2277.01    5573 2278.87  5593.3 2282.47    5644 2281.11
  5664.4 2289.61  5714.7 2297.65  5725.1 2301.09  5748.6  2303.7  5775.2 2306.63
    5786 2310.17  5840.8 2319.94  5896.2 2346.64  5907.7 2350.55  5929.5 2354.66
#Mann= 7 ,-1 , 0
    3883     .16       0  4024.2     .07       0  4982.8     .07       0
  4986.8     .07       0  5368.9     .16       0  5546.3    .035       0
  5748.6     .16       0
Bank Sta=4982.8,4986.8
XS Rating Curve= 0 ,0
Exp/Cntr=0.3,0.1

Type RM Length L Ch R = 1 ,28565   ,961,961,961
BEGIN DESCRIPTION:
Mapping XS 4071cbf3
END DESCRIPTION:
XS GIS Cut Line= 4
      1462070.88      6802674.38      1462960.65      6802683.06
       1463073.5      6802635.32      1463793.98      6802344.52
#Sta/Elev= 30
  4106.1 2288.23  4760.3 2271.37  4920.3 2264.03  4980.3 2258.39  5001.1 2259.06
  5033.2 2257.63  5054.9 2260.45  5087.5 2261.93    5125 2261.18  5141.6 2259.39
  5178.7 2259.46  5195.6  2257.2  5238.7 2261.45  5261.9 2260.46  5278.7 2256.57
  5278.9 2256.07  5282.7 2256.57  5339.8 2263.36    5388 2262.69  5393.4 2263.93
  5482.5 2266.35  5540.6 2268.59  5629.6 2274.87  5648.5  2276.7    5670 2281.44
  5715.5 2279.41    5724 2283.27  5787.9 2295.47  5819.4 2303.17  5895.4 2323.82
#Mann= 6 ,-1 , 0
  4106.1     .07       0  5278.7     .07       0  5282.7     .07       0
  5482.5     .16       0  5629.6    .035       0  5819.4     .16       0
#XS Ineff= 2 , 0
       0  5087.5 2261.93               0
Permanent Ineff=
       F       F
Bank Sta=5278.7,5282.7
XS Rating Curve= 0 ,0
Exp/Cntr=0.3,0.1

Type RM Length L Ch R = 1 ,27604   ,58,58,58
BEGIN DESCRIPTION:
Mapping XS 883ea3ff
END DESCRIPTION:
XS GIS Cut Line= 5
       1461908.2      6803268.53      1463100.75      6802983.76
       1463354.7      6803017.75      1463625.06      6802806.67
      1463917.45       6802422.6
#Sta/Elev= 30
  3517.7 2357.87  3606.9  2353.1  3637.8 2342.95  3672.2 2338.27  3699.5  2323.3
  3740.6 2310.33  3872.4  2301.4  3931.1 2296.66  4522.7 2272.63  4547.3 2271.76
  4696.7 2267.99  4741.4 2262.06  4798.5 2253.87  4891.6 2253.76  4959.5 2249.51
  4964.6  2251.7  5075.5 2245.86  5075.8 2245.36  5080.1 2245.86  5170.9 2250.39
  5214.3 2256.16  5313.8 2258.02  5349.4 2264.22  5466.4 2271.42  5499.1 2273.88
  5513.6 2278.89  5563.5 2276.98  5665.2 2302.99  5727.8 2314.86  5825.7 2353.12
#Mann= 10 ,-1 , 0
  3517.7     .07       0  3872.4    .035       0  3931.1     .07       0
  4522.7     .16       0  4547.3     .07       0  4741.4     .16       0
  5075.5     .07       0  5080.1     .16       0  5466.4    .035       0
  5665.2     .16       0
Bank Sta=5075.5,5080.1
XS Rating Curve= 0 ,0
Exp/Cntr=0.3,0.1

Type RM Length L Ch R = 1 ,27546   ,73,73,73
BEGIN DESCRIPTION:
Mapping XS 1db99b90
END DESCRIPTION:
XS GIS Cut Line= 5
      1462150.52      6803282.11       1463098.4      6803035.59
      1463320.62      6803066.84      1463428.26       6803059.9
      1463924.81      6802563.35
#Sta/Elev= 30
  3790.2 2310.34  3987.5 2296.88  4012.4 2295.68  4352.8 2279.58  4755.1 2266.24
  4822.3 2263.55  4827.3 2260.69  4887.4 2263.03  4898.6 2261.03  4947.9 2263.06
  5058.6  2261.2  5235.3 2263.19  5263.6 2261.63  5284.8 2256.99  5381.5 2256.48
  5381.8 2255.98  5386.1 2256.48  5419.1 2259.82  5433.3 2264.84  5528.7 2270.79
  5553.5 2272.47  5574.7 2278.03  5631.2 2277.04  5645.4 2282.37  5666.6 2284.57
  5714.9 2295.72  5751.5 2306.96  5779.7 2321.88  5800.7 2336.34  5804.1 2336.34
#Mann= 8 ,-1 , 0
  3790.2     .07       0  3987.5    .035       0  4012.4     .07       0
  4755.1     .16       0  5381.5     .07       0  5386.1     .16       0
  5528.7    .035       0  5714.9     .16       0
Bank Sta=5381.5,5386.1
XS Rating Curve= 0 ,0
Exp/Cntr=0.3,0.1

Type RM Length L Ch R = 1 ,27473   ,312,312,312
BEGIN DESCRIPTION:
Mapping XS f59f9656
END DESCRIPTION:
XS GIS Cut Line= 5
      1462118.12      6803376.12      1463093.81      6803094.87
      1463304.17      6803132.98      1463441.03      6803105.28
      1464003.15      6802702.78
#Sta/Elev= 30
  3770.8 2315.53  3849.9 2307.41    4017 2296.97  4127.6 2292.01  4759.5 2264.24
  4868.7 2257.56  4909.4  2254.3  4939.4 2249.62  5008.8 2244.94  5009.1 2244.44
  5013.4 2244.94  5041.7 2245.69  5104.4 2251.35  5427.4 2257.37  5455.4 2259.91
    5464 2263.39  5499.7 2264.12    5586 2270.45  5612.7 2272.36  5627.4 2276.18
    5663 2273.66  5677.8 2274.83  5692.5  2280.4  5734.9 2286.37  5763.8 2295.89
  5778.5 2304.56  5791.2 2307.47  5799.4 2309.49  5828.9 2323.12    5831 2327.67
#Mann= 8 ,-1 , 0
  3770.8     .07       0    4017    .035       0  4127.6     .07       0
  4759.5     .16       0  5008.8     .07       0  5013.4     .16       0
    5586    .035       0  5791.2     .16       0
Bank Sta=5008.8,5013.4
XS Rating Curve= 0 ,0
Exp/Cntr=0.3,0.1

Type RM Length L Ch R = 1 ,27161   ,340,340,340
BEGIN DESCRIPTION:
Mapping XS 39625050
END DESCRIPTION:
XS GIS Cut Line= 3
      1462361.74      6803598.85      1463485.82      6803373.17
      1464123.76      6802782.96
#Sta/Elev= 30
  3850.3 2293.52    3916 2290.07  4017.6 2285.06  4234.5 2279.28  4744.9 2259.08
  4841.6 2252.94  4892.5 2246.95  4914.4 2247.36  4943.4 2241.54  4987.4 2239.24
  4991.5 2239.17  4991.8 2238.67  4996.2 2239.17  5028.1 2245.32  5056.5 2248.06
  5184.1 2249.39  5339.4 2253.75  5481.2  2261.5  5502.1 2261.18  5581.3 2268.25
  5615.5 2272.78  5658.1 2271.55  5664.9 2273.28    5679 2281.43  5700.6 2284.18
  5805.5 2304.83  5827.6 2310.72    5835 2314.55  5855.9 2318.49  5865.9 2324.21
#Mann= 9 ,-1 , 0
  3850.3     .16       0    3916    .035       0  4017.6     .16       0
  4234.5     .07       0  4987.4     .16       0  4991.5     .07       0
  4996.2     .16       0  5581.3    .035       0  5805.5     .16       0
Bank Sta=4991.5,4996.2
XS Rating Curve= 0 ,0
Exp/Cntr=0.3,0.1

Type RM Length L Ch R = 1 ,26821   ,277,277,277
BEGIN DESCRIPTION:
Mapping XS 041c719e
END DESCRIPTION:
XS GIS Cut Line= 3
      1462528.98       6803896.7       1463636.6      6803657.12
      1464361.11      6803074.73
#Sta/Elev= 30
  3836.6 2283.51  3975.8 2278.47  4047.9 2273.69  4224.5  2267.7  4231.1 2267.54
  4421.3 2260.45  4436.2 2261.48  4465.4 2259.73  4470.5 2260.81  4563.8 2259.06
  4773.8 2252.64    4972  2242.9  5004.1 2236.26  5022.6 2235.41  5022.9 2234.91
  5027.3 2235.41  5053.7 2241.59  5074.5 2244.11  5118.8 2244.31  5266.5  2246.3
  5352.7 2250.78  5508.1 2253.76  5622.4 2259.25  5644.1 2261.74  5672.9  2261.5
  5700.1 2264.91  5743.3 2263.01  5757.7 2267.11  5864.7 2274.24  5899.4 2276.37
#Mann= 8 ,-1 , 0
  3836.6    .035       0  4224.5     .16       0  4231.1     .07       0
  5022.6     .07       0  5027.3     .07       0  5118.8     .16       0
  5622.4    .035       0  5864.7     .16       0
Bank Sta=5022.6,5027.3
XS Rating Curve= 0 ,0
Exp/Cntr=0.3,0.1

Type RM Length L Ch R = 1 ,26544   ,753,753,753
BEGIN DESCRIPTION:
Mapping XS e0448e5f
END DESCRIPTION:
XS GIS Cut Line= 3
      1462704.24      6804161.75      1463802.32      6803866.62
      1464539.13      6803082.13
#Sta/Elev= 30
  3858.7 2280.45  4056.2 2269.34  4248.5 2261.42  4377.7  2256.6  4651.8 2248.55
  4718.9 2245.43  4760.4  2246.1  4843.2 2243.14  4897.1 2235.28    4926  2234.8
  4957.1 2239.75  4992.1 2231.84  4992.4 2231.34    4997 2231.84  5010.7 2232.05
  5032.2 2237.99  5053.2  2239.2  5152.3  2239.5  5173.4 2240.26  5201.7 2244.15
    5255 2244.02  5336.4 2247.02  5562.6 2250.38  5661.4 2254.67  5725.3 2257.92
  5760.9 2262.17  5803.3 2260.01  5824.4  2263.5    5887 2266.18    6072 2276.42
#Mann= 9 ,-1 , 0
  3858.7     .16       0  4248.5     .07       0  4377.7     .16       0
  4651.8    .035       0  4992.1    .035       0    4997    .035       0
    5255     .16       0  5661.4    .035       0    5887     .16       0
Bank Sta=4992.1,4997
XS Rating Curve= 0 ,0
Exp/Cntr=0.3,0.1

Type RM Length L Ch R = 1 ,25791   ,508,508,508
BEGIN DESCRIPTION:
Mapping XS 39983ac3
END DESCRIPTION:
XS GIS Cut Line= 4
       1462717.2      6804647.87      1463954.23      6804530.68
      1464201.62      6804426.51      1465030.31      6803463.33
#Sta/Elev= 30
  3756.2 2282.72  3832.9 2275.48  3864.5 2271.11  3884.6 2272.78  4047.3 2259.79
  4121.7 2255.34    4629 2238.29  4728.7 2236.09  4818.7 2233.73    4866 2229.23
    4879 2231.15  4898.7  2227.6  4919.2 2223.87  4949.3 2225.52  4974.3 2223.47
  4994.2 2213.87  4994.5 2213.37  4999.1 2213.87  5010.5 2215.49  5017.2  2222.5
    5041 2228.23  5064.7 2229.44  5238.3 2227.56  5452.6 2230.49    5559 2235.15
  5665.5 2236.05  6080.2 2248.63  6400.4 2260.75  6453.7 2262.45  6537.8 2265.49
#Mann= 12 ,-1 , 0
  3756.2     .07       0  3832.9     .16       0  4047.3     .07       0
  4121.7     .16       0    4629     .07       0  4728.7    .035       0
  4898.7     .16       0  4994.2     .07       0  4999.1     .16       0
  6080.2    .035       0  6400.4     .07       0  6453.7     .16       0
Bank Sta=4994.2,4999.1
XS Rating Curve= 0 ,0
Exp/Cntr=0.3,0.1

Type RM Length L Ch R = 1 ,25283   ,621,621,621
BEGIN DESCRIPTION:
Mapping XS 81999447
END DESCRIPTION:
XS GIS Cut Line= 3
      1463387.36      6805353.61      1464181.66      6804936.93
       1465093.1      6803656.57
#Sta/Elev= 30
  3982.1    2252    4505 2234.61  4590.8 2232.32    4828  2226.2  4902.3 2223.95
  4966.1  2224.8  4980.9 2222.33  4995.6 2211.42  5007.8 2205.17  5008.2 2204.67
    5013 2205.17  5016.5  2205.6  5031.3 2214.97  5037.4 2216.54    5046 2221.13
  5060.8 2224.13  5173.9 2223.12  5454.7  2226.5  5798.4 2235.95  5820.7 2237.86
  6094.3 2247.26    6165 2250.24    6192 2249.15  6221.5 2251.13  6236.3 2250.96
  6242.4 2249.32    6251 2251.75  6326.9 2254.47  6420.6 2256.88  6450.7 2258.46
#Mann= 9 ,-1 , 0
  3982.1     .07       0    4505    .035       0  4590.8     .07       0
    4828     .16       0  5007.8     .07       0    5013     .16       0
  6094.3    .035       0  6326.9     .16       0  6420.6    .035       0
Bank Sta=5007.8,5013
XS Rating Curve= 0 ,0
Exp/Cntr=0.3,0.1

Type RM Length L Ch R = 1 ,24662   ,841,841,841
BEGIN DESCRIPTION:
Mapping XS 5982accd
END DESCRIPTION:
XS GIS Cut Line= 3
      1463403.88      6806061.06      1464788.43       6805084.5
      1465348.34      6803786.73
#Sta/Elev= 30
  3295.3 2250.73    3524 2236.65    3547  2235.6  3772.8 2227.88  4132.6 2225.36
  4246.8 2222.52  4264.7 2222.57  4428.4 2218.39  4491.1 2216.44  4605.2 2215.08
  4727.1 2217.75  4941.4 2216.11  4989.6 2207.98  5018.6 2199.67    5019 2199.17
  5024.2 2199.67  5039.4 2202.86  5051.1 2209.13  5073.8 2215.09  5144.4 2218.22
  5372.3 2221.05  5641.2 2230.47  5887.3 2236.32  5906.7 2236.28  6020.4 2238.67
  6074.2 2237.53  6085.8 2234.98  6103.2 2239.77    6175 2242.28    6403 2249.45
#Mann= 14 ,-1 , 0
  3295.3     .07       0    3524     .16       0    3547     .07       0
  4132.6     .16       0  4246.8     .07       0  4264.7     .16       0
  4428.4     .07       0  4491.1     .16       0  5018.6     .07       0
  5024.2     .16       0  5641.2    .035       0  5887.3     .16       0
  5906.7    .035       0    6175     .16       0
Bank Sta=5018.6,5024.2
XS Rating Curve= 0 ,0
Exp/Cntr=0.3,0.1

Type RM Length L Ch R = 1 ,23821   ,1058,1058,1058
BEGIN DESCRIPTION:
Mapping XS d8fb2305
END DESCRIPTION:
XS GIS Cut Line= 3
      1464135.99      6806028.55      1465394.68       6805603.2
      1465572.34      6805282.54
#Sta/Elev= 30
    3657 2213.67    3736 2212.39  3741.2 2213.74  3761.5 2211.73  3956.1 2209.83
    4036 2207.42  4194.3 2208.86  4384.3 2208.63  4454.1  2207.1  4686.8 2205.92
  4788.3  2204.9  4862.9 2202.89  4880.4 2201.85  4889.1  2199.4  4901.5 2201.72
  4912.1 2201.65  4920.6 2199.73  4925.8 2200.09  4943.7 2195.72  4957.3 2195.23
  4969.7 2192.82  4972.6    2192  4973.1  2191.5  4978.2    2192  4983.1 2195.73
  4991.2 2197.86  4996.9 2201.81  5018.7 2205.47  5161.1 2206.09  5352.2 2207.35
#Mann= 7 ,-1 , 0
    3657     .16       0  4686.8     .07       0  4788.3     .16       0
  4969.7     .16       0  4972.6     .07       0  4978.2     .16       0
  5161.1     .16       0
Bank Sta=4972.6,4978.2
XS Rating Curve= 0 ,0
Exp/Cntr=0.3,0.1

Type RM Length L Ch R = 1 ,22763   ,387,387,387
BEGIN DESCRIPTION:
Mapping XS 1d2f29e4
END DESCRIPTION:
XS GIS Cut Line= 3
      1464062.23      6806870.56      1465633.39      6806484.28
       1466040.5      6806003.54
#Sta/Elev= 30
  3408.6  2203.1  3526.9 2201.41  3576.2 2197.82    3771 2193.53  3975.8 2192.52
    4019 2192.52  4039.6 2190.94  4072.1 2191.17  4091.1 2192.29    4150 2191.12
  4223.5 2191.43  4286.8 2192.42  4861.3 2192.29  4874.3 2193.05  4902.9 2191.09
  4935.5 2184.37  4949.5 2184.34  4964.1 2182.81  4991.1 2184.27  5024.8 2187.85
  5032.5 2189.83  5067.6 2191.95  5223.6 2192.54  5237.9 2193.63  5258.8 2193.24
  5266.5 2194.07  5312.6 2193.55  5364.9 2194.12  5514.8 2196.48  5656.5 2195.57
#Mann= 8 ,-1 , 0
  3408.6     .07       0  3975.8    .035       0  4223.5     .07       0
  4874.3     .16       0  4949.5     .07       0  4991.1     .16       0
  5312.6     .07       0  5364.9     .16       0
#XS Ineff= 2 , 0
       0  4873.7    2193               0
Permanent Ineff=
       F       F
Bank Sta=4949.5,4991.1
XS Rating Curve= 0 ,0
Exp/Cntr=0.3,0.1

Type RM Length L Ch R = 1 ,22376   ,452,452,452
BEGIN DESCRIPTION:
Mapping XS ff691f20
END DESCRIPTION:
XS GIS Cut Line= 3
      1464517.96      6807504.23      1465880.79      6806749.03
       1466249.2      6806272.27
#Sta/Elev= 30
  3381.8 2198.01  3449.5 2194.22  3481.3 2194.49    3500 2193.29  3641.4 2186.96
  3728.6 2185.39  4083.7 2183.22  4148.9 2184.34  4289.7 2184.52  4376.7 2186.64
  4670.3 2186.93  4842.6 2185.99  4891.8  2186.2  4943.7 2184.61    4972 2181.91
  4979.1 2179.12  4986.5 2178.06  4992.9 2178.39  5004.5    2177    5005  2176.5
  5010.2    2177  5036.3 2183.57  5042.7 2184.01  5071.7 2183.45  5079.8 2185.47
  5206.6 2188.87  5378.7 2190.68    5443 2190.04  5513.6 2187.82  5542.4 2188.56
#Mann= 6 ,-1 , 0
  3381.8     .07       0    3500    .035       0  3728.6     .07       0
  4842.6     .16       0  5004.5     .07       0  5010.2     .16       0
#XS Ineff= 2 , 0
       0  4719.7    2189               0
Permanent Ineff=
       F       F
Bank Sta=5004.5,5010.2
XS Rating Curve= 0 ,0
Exp/Cntr=0.3,0.1

Type RM Length L Ch R = 1 ,21924   ,464,464,464
BEGIN DESCRIPTION:
Mapping XS 216ef0db
END DESCRIPTION:
XS GIS Cut Line= 3
       1465392.1      6807670.02      1466190.68      6807036.36
      1466389.75      6806642.56
#Sta/Elev= 30
  3970.6 2187.42  4002.1 2187.67  4080.6 2184.31  4109.5 2184.22  4159.1 2181.38
    4285 2179.75  4380.3  2177.7  4386.6 2175.68  4394.7 2175.63  4408.3 2177.37
  4421.9 2177.57  4522.9 2176.16  4614.2 2176.42  4628.6 2175.27  4771.2 2178.77
  4778.5 2178.05  4928.2 2178.37  4957.1 2177.81  4984.3 2174.08  5007.9 2174.26
  5010.6 2172.63  5011.1 2172.13  5016.3 2172.63  5044.2 2175.37  5066.6 2178.94
  5089.1 2180.17  5147.2 2180.53  5208.4 2182.38  5342.2 2184.38  5431.3 2184.52
#Mann= 4 ,-1 , 0
  3970.6     .07       0    4285     .16       0  5010.6     .07       0
  5016.3     .16       0
#XS Ineff= 2 , 0
       0  4771.2    2185               0
Permanent Ineff=
       F       F
Bank Sta=5010.6,5016.3
XS Rating Curve= 0 ,0
Exp/Cntr=0.3,0.1

Type RM Length L Ch R = 1 ,21460   ,420,420,420
BEGIN DESCRIPTION:
Mapping XS effe12d1
END DESCRIPTION:
XS GIS Cut Line= 4
      1465787.01      6807878.39      1466555.27      6807335.84
      1466616.03      6807123.17      1466464.33      6806672.41
#Sta/Elev= 30
    3958  2179.3  4178.7 2178.86  4208.3 2176.47  4237.1 2176.61  4273.5 2173.89
  4336.3 2173.82  4380.6 2171.65  4416.3 2172.39  4472.9 2169.87  4559.1 2169.56
  4631.7 2171.62    4739 2172.97  4811.6    2172  4861.5  2172.5  4913.8 2171.52
  4947.6 2170.23  4958.7 2168.59    4989 2167.86  4989.4 2167.36  4994.7 2167.86
  5064.6 2169.29  5093.2 2171.02  5188.5 2170.79    5229  2173.4  5265.8 2173.33
  5297.3 2175.72  5315.1 2175.68  5462.8 2181.64  5517.8    2183  5595.3 2183.06
#Mann= 4 ,-1 , 0
    3958     .07       0  4631.7     .16       0    4989     .07       0
  4994.7     .16       0
#XS Ineff= 2 , 0
       0    4739 2172.97               0
Permanent Ineff=
       F       F
Bank Sta=4989,4994.7
XS Rating Curve= 0 ,0
Exp/Cntr=0.3,0.1

Type RM Length L Ch R = 1 ,21040   ,706,706,706
BEGIN DESCRIPTION:
Mapping XS 8ed41b4c
END DESCRIPTION:
XS GIS Cut Line= 3
      1466364.29      6808290.71      1466983.22      6807216.05
      1466622.09      6806573.65
#Sta/Elev= 30
  3644.4 2171.83  3705.2 2171.74  3778.2 2169.21  3843.7 2168.04  3933.3 2168.52
    3998 2166.04  4028.3 2166.85  4051.1 2165.82    4334 2166.01  4409.2 2166.73
  4480.8 2165.86  4539.7  2166.7  4555.5 2165.93    4577 2166.71  4635.9 2166.83
  4716.4 2166.29  4759.5 2164.81  4775.3 2165.35  4861.5 2163.62  4936.8 2163.56
  4937.3 2163.06  4942.5 2163.56  5073.2 2166.03  5123.2 2170.09  5181.6 2171.12
  5256.8 2170.36  5402.8  2171.7  5580.7 2175.04  5586.4 2175.97  5621.5 2176.71
#Mann= 4 ,-1 , 0
  3644.4     .07       0    4334     .16       0  4936.8     .07       0
  4942.5     .16       0
#XS Ineff= 2 , 0
       0  4620.1    2170               0
Permanent Ineff=
       F       F
Bank Sta=4936.8,4942.5
XS Rating Curve= 0 ,0
Exp/Cntr=0.3,0.1

Type RM Length L Ch R = 1 ,20334   ,85,85,85
BEGIN DESCRIPTION:
Mapping XS f301ed00
END DESCRIPTION:
XS GIS Cut Line= 4
      1466805.49       6808399.3      1467218.67      6807552.11
      1467260.34      6807270.86      1467100.62      6806357.72
#Sta/Elev= 30
  4043.6 2164.75  4232.5 2165.69  4356.6 2161.93  4423.9 2162.19  4501.2 2158.76
  4553.5  2160.5  4765.8 2160.04  4852.6 2159.99  4902.6 2159.35  4942.1 2160.25
  4970.2 2157.87  4979.6 2155.75  4985.7 2152.14  4992.1 2151.48  4992.6 2150.98
  4998.6 2151.48  5010.5 2152.03  5030.8 2156.14    5051 2157.84  5203.8 2162.53
  5329.9 2164.48  5334.9  2163.7  5443.7 2164.84  5476.4 2163.94  5795.5  2166.9
  5914.5 2169.52  5968.9 2172.34  6028.4 2173.12  6075.4 2175.54  6197.5 2177.45
#Mann= 5 ,-1 , 0
  4043.6     .07       0  4765.8     .16       0  4852.6     .16       0
  4992.1     .07       0  4998.6     .16       0
Bank Sta=4992.1,4998.6
XS Rating Curve= 0 ,0
Exp/Cntr=0.3,0.1

Type RM Length L Ch R = 1 ,20249   ,115,115,115
BEGIN DESCRIPTION:
Mapping XS 79df8c98
END DESCRIPTION:
XS GIS Cut Line= 6
      1467012.92      6808470.55       1467280.3      6808328.15
      1467305.84      6807554.12      1467295.93      6807118.08
      1467257.73      6806517.39      1467162.79      6806252.54
#Sta/Elev= 30
  3906.4 2163.82  3940.4 2162.02  4002.4 2161.94  4078.7 2158.62  4160.1 2158.42
  4176.4 2156.67  4309.5 2156.94  4369.6 2155.53  4419.6 2155.82  4449.6  2157.5
  4769.8 2158.66  4839.8 2156.42  4879.9 2156.42  4976.1 2150.98  4976.6 2150.48
  4982.6 2150.98  4999.9 2151.16  5089.9 2158.45    5220 2162.59    5400 2165.78
  5730.7 2168.68  5827.2 2173.43  5832.2 2172.51  5981.1 2182.98  5986.4 2181.39
  6024.2 2183.51    6077 2181.48  6164.9 2181.04  6220.1 2182.33  6303.2 2179.96
#Mann= 6 ,-1 , 0
  3906.4     .07       0  4002.4     .16       0  4976.1     .07       0
  4982.6     .16       0  5986.4    .063       0  6164.9    .035       0
#XS Ineff= 2 , 0
       0  4769.8    2162               0
Permanent Ineff=
       F       F
Bank Sta=4976.1,4982.6
XS Rating Curve= 0 ,0
Exp/Cntr=0.3,0.1

Type RM Length L Ch R = 1 ,20134   ,366,366,366
BEGIN DESCRIPTION:
Mapping XS 15935705
END DESCRIPTION:
XS GIS Cut Line= 6
      1466839.69      6808945.61      1467416.95      6808489.88
      1467425.63      6807248.56      1467416.95       6806627.9
      1467403.93      6806432.59      1467440.42      6805912.34
#Sta/Elev= 30
  3325.3    2159  3629.4 2158.63  3768.4 2158.58  3811.8 2156.47  3911.1 2156.25
  3925.6 2153.64  3975.3 2154.71  4039.4 2152.12  4182.6 2153.04  4242.6 2150.64
  4302.6 2153.67  4521.4 2155.95    4847 2155.35  4872.6 2154.57  4892.6 2151.99
  4922.6 2152.52  4952.6 2150.56  4969.9 2149.37  4992.7 2150.71  5032.7 2156.79
  5102.7  2161.4  5462.8 2168.22  5792.8 2171.47  5822.8 2172.48  5852.8 2176.65
  6164.5 2185.91  6243.6 2186.69  6458.5 2184.44  6556.5 2190.84  6640.2 2193.22
#Mann= 9 ,-1 , 0
  3325.3     .07       0  3629.4     .07       0  4521.4     .16       0
    4847     .16       0  4952.6     .07       0  4992.7     .16       0
  6164.5    .035       0  6458.5     .16       0  6556.5     .07       0
#XS Ineff= 2 , 0
       0  4602.6    2162               0
Permanent Ineff=
       F       F
Bank Sta=4952.6,4992.7
XS Rating Curve= 0 ,0
Exp/Cntr=0.3,0.1

Type RM Length L Ch R = 1 ,19768   ,752,752,752
BEGIN DESCRIPTION:
Mapping XS f8867216
END DESCRIPTION:
XS GIS Cut Line= 5
      1466974.56      6808973.36      1467429.39      6808594.92
      1467634.25       6807834.5       1468415.5      6807275.47
      1468730.75      6807150.76
#Sta/Elev= 30
  3608.6 2155.83  3742.3 2156.09  4017.3 2155.65  4038.5 2154.73    4046 2152.59
  4095.4 2153.56    4167 2150.51  4252.5 2150.99  4342.1 2151.04  4391.8 2147.66
  4424.9 2151.61  4471.6 2152.82  4699.9 2153.84  4890.2 2152.15  4935.3 2148.35
  4983.4 2148.24  4987.4 2146.69  4987.9 2146.19  4997.8 2146.69    5043 2153.61
  5109.1 2155.53  5265.4 2158.72  5394.5 2155.92  5428.2 2157.54  5493.9  2162.4
  5670.4 2165.62  5932.5 2172.61  6139.8  2172.5  6254.5 2174.86  6287.5 2175.04
#Mann= 11 ,-1 , 0
  3608.6     .07       0  3742.3    .035       0  4252.5     .07       0
  4699.9     .16       0  4987.4     .07       0  4997.8     .16       0
  5109.1    .035       0  5428.2     .16       0  5670.4     .07       0
  6139.8     .16       0  6254.5     .07       0
#XS Ineff= 2 , 0
       0    4661    2156               0
Permanent Ineff=
       F       F
Bank Sta=4987.4,4997.8
XS Rating Curve= 0 ,0
Exp/Cntr=0.3,0.1

Type RM Length L Ch R = 1 ,19016   ,467,467,467
BEGIN DESCRIPTION:
Mapping XS fc974419
END DESCRIPTION:
XS GIS Cut Line= 3
      1466871.38      6809177.05      1467652.67      6808508.62
      1468329.78      6808478.23
#Sta/Elev= 30
  3782.2 2157.35  3819.5 2158.23  3960.7 2155.48  4003.9 2156.27  4052.1 2154.06
  4358.5 2153.78    4366 2151.33  4407.9 2152.52  4479.3 2149.35  4533.2 2149.78
  4635.1 2149.67  4677.9 2145.94  4713.1 2147.54  4727.3 2146.23  4748.2 2140.75
  4776.7 2148.16  4805.3 2149.23  4862.8 2148.65  4906.6 2144.76  4967.2 2137.03
  4977.6  2131.8  4978.1  2131.3  4988.2  2131.8    5043 2147.13  5144.7 2152.83
  5168.9 2154.09  5263.2 2158.12  5313.2 2157.26  5370.3 2159.28  5488.2 2159.75
#Mann= 11 ,-1 , 0
  3782.2    .035       0  3960.7     .07       0  4052.1    .035       0
  4533.2     .07       0  4906.6     .16       0  4967.2     .16       0
  4977.6     .07       0  4988.2     .16       0  5144.7     .16       0
  5168.9     .07       0  5370.3    .045       0
#XS Ineff= 2 , 0
       0  4805.3 2149.23               0
Permanent Ineff=
       F       F
Bank Sta=4977.6,4988.2
XS Rating Curve= 0 ,0
Exp/Cntr=0.3,0.1

Type RM Length L Ch R = 1 ,18549   ,212,212,212
BEGIN DESCRIPTION:
Mapping XS cfa30e48
END DESCRIPTION:
XS GIS Cut Line= 3
       1466885.3      6809207.41      1467268.12      6808941.78
      1468395.72      6808960.01
#Sta/Elev= 30
  3983.7 2156.38    4083 2155.25  4127.5 2156.17  4285.6 2152.33  4312.6 2153.58
  4448.6 2152.79  4476.5 2151.96  4496.5 2149.81  4528.4 2150.92  4621.8 2146.34
  4696.6 2142.29  4776.6 2145.14  4880.2 2144.63  4896.6 2144.58  4926.6 2141.52
  4956.6 2136.04  4976.6  2134.3  4986.6 2132.39    4991 2126.96  4991.5 2126.46
  5002.2 2126.96  5056.6 2138.63  5076.6 2140.26  5096.6 2143.99  5116.6 2146.04
  5229.8 2146.65  5276.6 2147.58  5316.6 2150.31  5454.5 2150.87  5577.4  2152.6
#Mann= 7 ,-1 , 0
  3983.7    .035       0  4621.8     .07       0  4880.2     .16       0
    4991     .07       0  5002.2     .16       0  5229.8     .07       0
  5454.5    .045       0
Bank Sta=4991,5002.2
XS Rating Curve= 0 ,0
Exp/Cntr=0.3,0.1

Type RM Length L Ch R = 1 ,18337   ,473,473,473
BEGIN DESCRIPTION:
Mapping XS 4d6c8fa5
END DESCRIPTION:
XS GIS Cut Line= 4
      1466903.57       6809345.4      1467171.76      6809165.74
      1467838.43      6809147.51      1468416.53      6809168.34
#Sta/Elev= 30
  4004.6 2153.96  4109.3 2154.05  4205.7  2152.7  4262.8 2153.69  4350.7 2150.21
  4431.6 2150.17  4470.7 2148.22  4500.7 2148.99  4594.6 2141.95  4620.8 2139.23
  4670.8 2137.71  4722.4 2139.96  4794.6    2143  4850.8 2142.57  4890.9 2135.12
  4970.9 2132.65  4990.1 2128.66  5015.3 2126.37  5015.8 2125.87  5026.5 2126.37
  5030.9 2127.31  5040.9 2135.15  5050.9 2140.58  5060.9 2142.42  5193.2  2143.6
  5241.1 2145.64    5398 2146.56  5504.6 2148.96  5517.7 2149.06  5572.8 2149.29
#Mann= 10 ,-1 , 0
  4004.6     .07       0  4109.3    .035       0  4594.6     .07       0
  4722.4     .16       0  5015.3     .07       0  5026.5     .16       0
  5193.2     .07       0    5398    .045       0  5504.6     .07       0
  5517.7    .045       0
Bank Sta=5015.3,5026.5
XS Rating Curve= 0 ,0
Exp/Cntr=0.3,0.1

Type RM Length L Ch R = 1 ,17864   ,440,440,440
BEGIN DESCRIPTION:
Mapping XS f1eef065
END DESCRIPTION:
XS GIS Cut Line= 3
      1467064.09      6809545.94      1467642.25      6809553.76
      1468428.72      6809548.55
#Sta/Elev= 30
  4408.9 2150.24  4509.3 2149.85  4639.8 2147.92  4659.8 2146.22  4689.8  2147.4
  4729.8 2142.62  4781.1 2141.15  4789.8 2141.47  4809.8 2138.84  4829.8 2131.65
  4839.8 2129.87  4878.2 2129.15  4899.9 2131.47    4928 2132.17  4959.9 2129.02
  4969.9 2126.88  4980.4 2122.43  4980.9 2121.93  4991.6 2122.43  4999.9 2126.61
  5029.9 2128.26  5079.9 2137.79  5129.9 2139.64  5259.9 2139.26  5433.8 2135.99
  5545.7    2140  5566.5 2141.02  5579.9 2142.48  5740.3 2143.11  5773.6 2143.52
#Mann= 10 ,-1 , 0
  4408.9     .07       0  4509.3    .035       0  4781.1     .07       0
  4878.2     .16       0  4980.4     .07       0  4991.6     .16       0
  5433.8     .07       0  5545.7    .045       0  5566.5     .07       0
  5740.3    .045       0
Bank Sta=4980.4,4991.6
XS Rating Curve= 0 ,0
Exp/Cntr=0.3,0.1

Type RM Length L Ch R = 1 ,17424   ,654,654,654
BEGIN DESCRIPTION:
Mapping XS fb41d052
END DESCRIPTION:
XS GIS Cut Line= 3
      1467316.69      6810194.41      1467655.27      6809960.01
      1468430.64      6809606.15
#Sta/Elev= 30
  4571.6 2142.54  4595.8 2144.39  4712.4 2143.66  4783.6 2143.44  4834.3 2139.29
  4855.3 2139.56  4870.1  2137.9  4923.1 2135.88  4947.8 2133.05  4962.7 2129.53
  4980.8 2120.42    4986 2120.42  4988.4 2118.64  4988.9 2118.14  4999.7 2118.64
  4999.9 2121.64  5005.4 2123.67  5051.5 2125.91  5189.7 2124.48  5212.7  2125.4
  5269.8 2130.44  5287.3 2130.24  5338.9 2132.75    5385 2131.07  5413.5 2131.97
  5497.4 2131.22  5565.7 2133.88  5654.9 2140.46  5714.1 2140.82  5835.7 2142.12
#Mann= 7 ,-1 , 0
  4571.6    .035       0  4712.4     .07       0  4923.1     .16       0
  4988.4     .07       0  4999.7     .16       0  5497.4     .07       0
  5714.1    .045       0
Bank Sta=4988.4,4999.7
XS Rating Curve= 0 ,0
Exp/Cntr=0.3,0.1

Type RM Length L Ch R = 1 ,16770   ,569,569,569
BEGIN DESCRIPTION:
Mapping XS db3f54b0
END DESCRIPTION:
XS GIS Cut Line= 3
      1467672.65      6810671.79       1468214.3      6810059.83
      1468435.65      6809718.69
#Sta/Elev= 30
  4173.2 2132.26  4460.6 2131.54  4652.2 2132.25  4666.4  2133.2  4694.8 2130.65
  4751.7  2127.9  4758.4 2127.37  4772.6 2124.54  4801.1 2122.61  4872.2 2120.28
  4899.7 2120.95  4919.1 2120.47  4956.6 2118.51  4994.5 2118.63  5005.7 2119.42
  5015.2  2115.7  5015.7  2115.2  5026.6  2115.7    5042 2119.97  5051.1 2123.63
  5057.1 2124.61  5064.1 2127.48  5118.9 2132.05  5150.7 2135.35  5202.1 2137.17
  5217.3 2138.07    5231 2139.97    5308 2139.79  5347.1 2140.08  5397.1 2141.88
#Mann= 6 ,-1 , 0
  4173.2     .07       0  4919.1     .16       0  5015.2     .07       0
  5026.6     .16       0  5118.9     .07       0    5308    .045       0
Bank Sta=5015.2,5026.6
XS Rating Curve= 0 ,0
Exp/Cntr=0.3,0.1

Type RM Length L Ch R = 1 ,16201   ,330,330,330
BEGIN DESCRIPTION:
Mapping XS 25ed8b0d
END DESCRIPTION:
XS GIS Cut Line= 3
      1468080.63      6810947.19      1468563.26      6810464.56
      1468917.44       6810106.9
#Sta/Elev= 30
  4339.8 2127.78  4752.4 2127.74  4823.2  2126.7  4844.4 2128.34  4929.2 2123.17
  4971.6 2119.32  4992.9 2114.39  5001.3 2110.67  5001.8 2110.17  5012.7 2110.67
  5014.1 2112.82  5022.3 2113.02  5028.2 2115.34  5042.4 2113.52  5063.6 2115.89
  5091.1 2116.22    5106 2119.77  5113.1 2122.91  5120.1 2123.18  5127.2 2125.75
  5141.4 2127.92  5155.5 2128.14  5176.7 2125.95  5212.1  2129.5  5235.6 2129.23
  5275.7 2130.33  5311.1 2134.83  5347.5 2134.21  5417.6 2135.07  5525.7 2136.25
#Mann= 7 ,-1 , 0
  4339.8     .07       0  5001.3     .07       0  5012.7     .07       0
  5091.1     .16       0  5235.6    .045       0  5347.5     .16       0
  5417.6    .045       0
Bank Sta=5001.3,5012.7
XS Rating Curve= 0 ,0
Exp/Cntr=0.3,0.1

Type RM Length L Ch R = 1 ,15871   ,437,437,437
BEGIN DESCRIPTION:
Mapping XS 01d91fe5
END DESCRIPTION:
XS GIS Cut Line= 3
      1468301.29      6811110.39      1468861.17      6810537.48
       1469068.7      6810322.17
#Sta/Elev= 30
  4211.7 2125.66  4247.8  2125.6    4513 2124.76    4605 2125.24  4640.3 2123.76
  4696.9 2124.07  4760.4 2118.71  4795.9 2116.97    4810 2116.88    4817 2115.94
  4866.6 2113.46  4888.3 2113.02    4916 2112.47  4951.5 2113.32  4965.6 2112.75
  4979.8 2110.85  4995.2 2110.06  4995.7 2109.56  5006.1 2109.56  5006.6 2110.06
  5008.1 2113.87  5011.6 2117.32  5015.9 2117.62  5022.2 2121.35  5036.4 2124.85
  5071.6  2127.4    5093 2129.82  5141.6 2129.83  5206.2 2133.25  5311.8  2132.9
#Mann= 7 ,-1 , 0
  4211.7    .035       0  4247.8     .07       0  4888.3     .16       0
  4995.2     .07       0  5006.6     .16       0  5011.6     .07       0
  5141.6    .045       0
Bank Sta=4995.2,5006.6
XS Rating Curve= 0 ,0
Exp/Cntr=0.3,0.1

Type RM Length L Ch R = 1 ,15434   ,625,625,625
BEGIN DESCRIPTION:
Mapping XS 753c28c1
END DESCRIPTION:
XS GIS Cut Line= 3
      1468642.41      6811274.47      1469030.44      6810928.11
      1469225.73      6810688.56
#Sta/Elev= 30
  4469.5 2122.31  4638.7 2121.79  4681.3  2120.9  4752.4 2120.77  4808.4 2119.41
  4865.3 2119.49  4915.3 2114.32  4936.3  2113.5  4957.2  2110.3    4979 2108.84
  4994.8 2106.86  4995.3 2106.36  5005.7 2106.36  5006.2 2106.86  5006.9 2107.49
  5014.9  2107.7  5035.7 2109.95  5056.5 2110.82  5064.4 2112.34  5078.8  2113.6
  5099.6 2114.63    5106 2116.15  5113.9 2115.65  5120.4 2116.68  5184.3 2122.55
  5256.1 2126.24  5284.8 2129.79  5291.3 2129.73  5295.9 2131.06  5298.7 2131.06
#Mann= 3 ,-1 , 0
  4469.5     .07       0  4994.8     .07       0  5006.2     .07       0
Bank Sta=4994.8,5006.2
XS Rating Curve= 0 ,0
Exp/Cntr=0.3,0.1

Type RM Length L Ch R = 1 ,14809   ,323,323,323
BEGIN DESCRIPTION:
Mapping XS e7473531
END DESCRIPTION:
XS GIS Cut Line= 3
      1469125.03      6811788.96      1469494.85      6811348.82
      1469557.35       6810835.8
#Sta/Elev= 30
  4406.5 2117.14  4442.9 2115.69  4463.7 2116.11  4471.5 2117.12  4506.6 2116.39
  4577.8 2116.78  4662.7 2116.98  4726.4  2115.7  4783.7 2116.45  4917.7 2115.71
    4932 2113.75  4946.3  2108.2  4952.9 2106.84  4960.6 2104.96    4973 2103.52
  4973.5 2103.02  4984.4 2103.52  5052.7  2105.4    5093 2105.46  5133.3  2108.1
  5194.1 2109.74  5270.7 2114.69  5287.6  2114.3  5304.6 2116.82  5352.3 2115.34
    5363 2116.24  5445.6 2117.26  5465.8 2120.38  5485.9  2120.9  5498.2 2119.52
#Mann= 7 ,-1 , 0
  4406.5    .035       0  4577.8     .07       0  4952.9     .16       0
    4973     .07       0  4984.4     .16       0  5287.6     .07       0
    5363     .16       0
Bank Sta=4973,4984.4
XS Rating Curve= 0 ,0
Exp/Cntr=0.3,0.1

Type RM Length L Ch R = 1 ,14486   ,186,186,186
BEGIN DESCRIPTION:
Mapping XS 49ff7480
END DESCRIPTION:
XS GIS Cut Line= 3
      1469619.83      6811781.16      1469796.94      6811403.51
      1469604.23      6810786.31
#Sta/Elev= 30
    4464 2114.63  4491.5 2112.84  4508.8 2114.08  4601.8  2113.4  4787.8 2113.32
  4816.5 2110.51  4822.1 2111.04  4921.4 2104.69    4936 2103.25  4941.2 2103.55
  4973.7 2101.43    5001 2099.12  5017.3 2096.84  5017.8 2096.34  5028.8 2096.84
  5038.7 2098.98    5044 2101.23    5065 2105.72  5103.7 2106.24  5174.4 2109.37
  5244.1 2113.19    5264 2113.23    5285 2114.72  5352.2 2116.16  5406.6 2115.85
  5452.6 2117.43  5471.5 2117.08    5504 2118.16  5509.3 2119.08  5527.7 2118.84
#Mann= 7 ,-1 , 0
    4464    .035       0  4601.8     .07       0  4921.4     .16       0
  5017.3     .07       0  5028.8     .16       0  5174.4     .07       0
  5352.2     .16       0
Bank Sta=5017.3,5028.8
XS Rating Curve= 0 ,0
Exp/Cntr=0.3,0.1

Type RM Length L Ch R = 1 ,14300   ,314,314,314
BEGIN DESCRIPTION:
Mapping XS 2098289b
END DESCRIPTION:
XS GIS Cut Line= 3
      1469742.23      6811796.78      1469934.96      6811320.18
       1469898.5      6810528.51
#Sta/Elev= 30
  4403.2 2113.12    4421 2113.57    4445 2111.81  4466.6 2112.77    4555 2112.16
  4736.3 2112.67  4856.4 2105.01  4949.5  2100.1  4973.6 2097.48  4974.1 2096.98
  4985.4 2097.48  5019.6  2101.4  5025.4 2100.64  5029.8 2099.01  5059.6 2099.55
  5069.6 2101.13  5099.7 2102.48  5159.7 2104.19  5179.8 2103.12  5199.8 2105.28
  5276.8 2106.85  5329.9 2108.77    5410 2108.65    5440 2110.18  5457.4 2112.73
  5470.1 2112.02  5490.1  2113.1  5510.1 2115.92  5571.3 2117.79  5709.8 2120.79
#Mann= 8 ,-1 , 0
  4403.2    .035       0    4555     .07       0  4856.4     .16       0
  4973.6     .07       0  4985.4     .16       0  5025.4     .07       0
  5276.8    .035       0  5571.3     .16       0
Bank Sta=4973.6,4985.4
XS Rating Curve= 0 ,0
Exp/Cntr=0.3,0.1

Type RM Length L Ch R = 1 ,13986   ,383,383,383
BEGIN DESCRIPTION:
Mapping XS 34cd6b37
END DESCRIPTION:
XS GIS Cut Line= 4
      1469808.45      6811790.64      1469873.54      6811681.29
      1470183.44      6811394.83      1470446.46      6810978.17
#Sta/Elev= 30
  4430.1 2113.17  4473.1 2111.11  4488.7 2112.52  4552.9 2111.43  4595.1 2111.86
  4631.4  2112.2  4667.1 2110.73  4737.4    2110  4794.1 2108.25  4850.8    2108
  4921.5 2103.74  4981.6  2099.5  4999.3 2097.78    5017 2093.56  5017.5 2093.06
  5028.9 2093.56  5050.2 2095.92  5071.4 2103.33  5080.7 2103.67  5093.9  2105.6
  5138.4  2103.7  5188.5 2103.71  5311.4 2108.64    5342 2112.92  5347.9 2113.04
    5354 2117.71  5373.3 2121.93  5384.3 2123.74  5420.8 2125.87  5472.1 2127.12
#Mann= 7 ,-1 , 0
  4430.1    .035       0  4595.1     .07       0  4921.5     .16       0
  4981.6     .07       0    5017     .07       0  5028.9     .07       0
  5373.3     .16       0
Bank Sta=5017,5028.9
XS Rating Curve= 0 ,0
Exp/Cntr=0.3,0.1

Type RM Length L Ch R = 1 ,13603   ,247,247,247
BEGIN DESCRIPTION:
Mapping XS 59fe925b
END DESCRIPTION:
XS GIS Cut Line= 4
      1469831.89      6811788.04      1469909.03      6811693.37
      1470311.04      6811678.68      1470945.52      6811682.95
#Sta/Elev= 30
  4480.7 2112.76  4496.8 2112.78  4519.1 2110.82  4525.6 2110.78  4532.3 2112.07
  4613.4 2112.06    4839 2107.46    4899 2108.05  4907.7 2106.11    4969 2100.47
  4999.1 2095.79  5004.6 2091.97  5009.6 2091.97  5013.1 2088.68  5013.6 2088.18
  5025.1 2088.68  5029.1 2090.58  5059.1 2095.01  5089.1 2095.91  5204.7 2103.68
  5249.1 2105.84  5309.1 2107.18  5339.1 2109.82  5359.1 2112.75  5389.1 2112.13
  5409.1 2115.75  5439.1 2117.16  5459.1 2116.11  5589.1 2120.31  5639.6 2120.36
#Mann= 5 ,-1 , 0
  4480.7    .035       0  4907.7    .094       0  5013.1     .07       0
  5025.1    .094       0  5204.7    .035       0
Bank Sta=5013.1,5025.1
XS Rating Curve= 0 ,0
Exp/Cntr=0.3,0.1

Type RM Length L Ch R = 1 ,13356   ,196,196,196
BEGIN DESCRIPTION:
Mapping XS 10b6ceb0
END DESCRIPTION:
XS GIS Cut Line= 3
      1469767.18      6811898.23      1470381.77      6811887.81
      1470904.16      6811893.01
#Sta/Elev= 30
  4366.6 2111.66  4564.5 2109.92  4614.5 2110.73  4634.5 2109.43  4672.3 2108.51
  4754.5 2107.77  4807.2 2104.45  4834.5 2103.75  4904.5 2097.86  4934.5  2094.6
  4954.5 2093.79  4964.5 2090.57  4974.4  2085.3  4974.9  2084.8  4986.4  2085.3
  4994.5 2087.93  5014.5 2099.99  5024.5  2104.2  5044.5 2106.22  5104.5 2106.62
  5124.5 2107.91  5144.5 2111.17  5154.5 2111.83  5244.5 2115.38  5294.5 2118.18
  5334.5 2121.77  5364.5 2126.06  5454.5 2129.43  5501.1 2129.37  5503.7  2130.1
#Mann= 4 ,-1 , 0
  4366.6    .035       0  4807.2     .16       0  4974.4     .07       0
  4986.4     .16       0
Bank Sta=4974.4,4986.4
XS Rating Curve= 0 ,0
Exp/Cntr=0.3,0.1

Type RM Length L Ch R = 1 ,13160   ,359,359,359
BEGIN DESCRIPTION:
Mapping XS 24375ab3
END DESCRIPTION:
XS GIS Cut Line= 3
      1469798.45       6812195.1      1470324.48       6812064.9
      1470880.88       6812132.5
#Sta/Elev= 30
  4427.1 2109.07  4644.1 2108.65  4680.8 2107.43  4753.2 2107.77  4842.8 2103.43
  4876.8 2102.33    4893 2099.93  4898.1 2100.54  4928.3  2097.4  4966.7 2090.58
  4971.8 2090.58  4979.6 2087.84  4983.7 2083.46  4984.2 2082.96  4995.7 2083.46
  5019.9 2091.42  5035.6 2093.85  5040.6 2093.29  5060.2 2096.29  5090.4 2098.45
  5150.9 2105.82  5181.1  2108.2  5204.1 2107.72  5271.7 2118.47  5280.9 2119.54
  5285.9  2118.4    5312 2125.95  5322.1 2127.16  5382.5 2130.82  5529.5  2131.9
#Mann= 5 ,-1 , 0
  4427.1     .07       0  4644.1    .035       0  4842.8     .16       0
  4983.7     .07       0  4995.7     .16       0
Bank Sta=4983.7,4995.7
XS Rating Curve= 0 ,0
Exp/Cntr=0.3,0.1

Type RM Length L Ch R = 1 ,12801   ,336,336,336
BEGIN DESCRIPTION:
Mapping XS 275bf89d
END DESCRIPTION:
XS GIS Cut Line= 3
        1469926.      6812544.08       1470337.5      6812395.63
      1470756.75        6812380.
#Sta/Elev= 30
  4545.1 2104.75  4640.9 2105.48  4671.6 2104.17    4746 2104.66  4780.8 2102.82
  4826.8 2101.86  4852.3 2099.97  4884.2 2100.61    4901 2097.97  4934.1 2096.81
  4962.4 2094.59  4969.3 2089.68  4978.6 2084.85  4982.6 2084.85  4994.1 2081.68
  4994.6 2081.18  5006.1 2081.68  5010.1 2085.96  5020.1 2089.11  5090.1 2091.79
  5240.2 2104.13  5260.3 2108.14  5270.3 2112.65  5300.3 2123.12  5310.3 2124.37
  5323.4 2123.76  5350.3 2125.93  5370.3 2126.51  5380.3 2128.16  5402.1 2129.42
#Mann= 6 ,-1 , 0
  4545.1     .07       0  4780.8    .035       0  4826.8     .07       0
  4934.1     .16       0  4994.1     .07       0  5006.1     .16       0
Bank Sta=4994.1,5006.1
XS Rating Curve= 0 ,0
Exp/Cntr=0.3,0.1

Type RM Length L Ch R = 1 ,12465   ,264,264,264
BEGIN DESCRIPTION:
Mapping XS cd60cbb6
END DESCRIPTION:
XS GIS Cut Line= 3
      1470072.27      6812831.73      1470444.62      6812685.91
      1470944.65      6812573.92
#Sta/Elev= 30
  4586.7 2101.64  4623.5 2101.96  4670.9 2101.95  4776.4 2099.82  4830.6 2100.22
  4879.6 2096.43  4922.6 2091.61  4939.2 2088.89    4969 2088.17  4984.1 2084.06
  4989.3 2084.06  4995.1 2079.34  4995.6 2078.84  5007.2 2079.34  5007.5 2082.31
  5017.7 2086.54    5048 2087.25    5069 2087.62  5141.5 2092.09  5161.2 2092.19
  5179.7 2093.95  5228.2 2095.22  5233.4 2096.19  5253.4 2095.73  5271.6 2096.98
  5314.9 2097.53  5427.6 2103.36  5448.1 2103.36  5460.5 2104.45    5499 2105.63
#Mann= 6 ,-1 , 0
  4586.7     .07       0  4623.5    .035       0  4670.9     .07       0
  4995.1     .07       0  5007.2     .07       0    5048     .16       0
Bank Sta=4995.1,5007.2
XS Rating Curve= 0 ,0
Exp/Cntr=0.3,0.1

Type RM Length L Ch R = 1 ,12201   ,354,354,354
BEGIN DESCRIPTION:
Mapping XS 078acb9c
END DESCRIPTION:
XS GIS Cut Line= 3
      1470224.68      6813219.79      1470600.14      6812896.41
      1470984.28      6812716.28
#Sta/Elev= 30
  4501.6 2098.51  4588.2 2098.11  4637.6 2098.66  4729.8 2098.08  4786.8 2096.81
  4858.1 2096.89  4899.8 2092.99  4907.5 2092.83  4914.1 2090.12  4921.7  2090.2
  4928.3 2086.35  4950.3 2080.31  4963.9  2079.1  4971.1 2077.79  4971.7 2076.82
  4972.2 2076.32  4983.3 2076.32  4983.8 2076.82    4992 2080.36    4997 2084.17
  5031.5 2085.29  5052.2 2085.82  5057.8 2085.28  5075.1 2086.91  5097.9  2086.7
  5157.1 2088.36  5314.3 2098.21  5354.4  2099.6    5367 2101.16  5421.4 2103.53
#Mann= 4 ,-1 , 0
  4501.6     .07       0  4971.7     .07       0  4983.8     .07       0
  5031.5     .16       0
Bank Sta=4971.7,4983.8
XS Rating Curve= 0 ,0
Exp/Cntr=0.3,0.1

Type RM Length L Ch R = 1 ,11847   ,404,404,404
BEGIN DESCRIPTION:
Mapping XS 1809dde6
END DESCRIPTION:
XS GIS Cut Line= 3
       1470259.4      6813415.09      1470791.11       6813180.7
      1471107.96       6812846.5
#Sta/Elev= 30
  4414.4 2096.79  4521.5 2096.79  4718.6 2095.41  4759.3 2095.34  4864.5 2092.55
  4927.7 2092.01  4968.7 2092.05  4977.9 2090.89    4992 2087.72  4994.9    2085
  5000.8    2085  5014.1 2078.35  5015.3 2075.97  5015.8 2075.47  5027.4 2075.97
  5035.6 2077.08  5049.7    2082  5084.9 2082.32  5099.1 2083.32  5131.7 2083.15
  5155.7 2083.93  5198.2  2087.4  5212.3 2087.44  5247.5 2090.67  5339.7 2095.85
  5360.8 2095.35  5368.1 2094.51  5401.3 2096.86  5410.5 2097.61    5456 2097.27
#Mann= 7 ,-1 , 0
  4414.4     .07       0  4718.6    .035       0  4927.7     .07       0
  5015.3     .07       0  5027.4     .07       0  5131.7     .16       0
  5401.3    .035       0
Bank Sta=5015.3,5027.4
XS Rating Curve= 0 ,0
Exp/Cntr=0.3,0.1
