--- MULBERRY CREEK TRIBUTARY 4.prj (project) ---

Proj Title=MULBERRY CREEK TRIBUTARY 4 Base Level Engineering
Current Plan=p01
Default Exp/Contr=0.3,0.1
English Units
Geom File=g01
Flow File=f01
Plan File=p01
Y Axis Title=Elevation
X Axis Title(PF)=Main Channel Distance
X Axis Title(XS)=Station
BEGIN DESCRIPTION:
MULBERRY CREEK TRIBUTARY 4
END DESCRIPTION:
DSS Export Rating Curves= 0
DSS Export Rating Curve Sorted= 0
DSS Export Volume Flow Curves= 0
DXF OffsetX= 0
DXF OffsetY= 0
DXF ScaleX= 1
DXF ScaleY= 10

--- MULBERRY CREEK TRIBUTARY 4.p01 (plan) ---

Plan Title=Multiple Run
Short Identifier=Multiple
Geom File=g01
Flow File=f01
Subcritical Flow
K Sum by GR= 0
Std Step Tol= 0.01
Critical Tol= 0.01
Num of Std Step Trials= 20
Max Error Tol= 0.3
Flow Tol Ratio= 0.001
Split Flow NTrial= 30
Split Flow Tol= 0.02
Split Flow Ratio= 0.02
Log Output Level= 0
Friction Slope Method= 1
Unsteady Friction Slope Method= 2
Unsteady Bridges Friction Slope Method= 1
Parabolic Critical Depth
Global Vel Dist=  1 , 1 , 1
Global Log Level= 0
CheckData=True
Encroach Param= -1, 0, 0, 0
BEGIN DESCRIPTION:
Multiple Run
END DESCRIPTION:

--- MULBERRY CREEK TRIBUTARY 4.f01 (steady flow) ---

Flow Title=Multiple
Program Version=4.10
Number of Profiles= 7
Profile Names=10-year,25-year,50-year,1pct_min,100-year,1pct_plu,500-year
River Rch & RM=MULBERRY CREEK T,Reach-1         ,35439
     175     237     286     173     345     688     506
River Rch & RM=MULBERRY CREEK T,Reach-1         ,29335
     354     499     620     384     765    1527    1181
River Rch & RM=MULBERRY CREEK T,Reach-1         ,23553
     458     653     819     510    1018    2030    1594
River Rch & RM=MULBERRY CREEK T,Reach-1         ,20201
     483     690     865     539    1076    2146    1686
River Rch & RM=MULBERRY CREEK T,Reach-1         ,16169
     585     842    1063     666    1329    2652    2107
River Rch & RM=MULBERRY CREEK T,Reach-1         ,14581
     588     846    1067     668    1332    2658    2107
River Rch & RM=MULBERRY CREEK T,Reach-1         ,12347
     680     985    1247     784    1564    3120    2493
River Rch & RM=MULBERRY CREEK T,Reach-1         ,9777
     732    1061    1345     845    1686    3364    2689
River Rch & RM=MULBERRY CREEK T,Reach-1         ,5391
     761    1103    1397     877    1751    3493    2790
Boundary for River Rch & Prof#=MULBERRY CREEK T,Reach-1         , 1
Up Type= 0
Dn Type= 3
Dn Slope=0.005
Boundary for River Rch & Prof#=MULBERRY CREEK T,Reach-1         , 2
Up Type= 0
Dn Type= 3
Dn Slope=0.005
Boundary for River Rch & Prof#=MULBERRY CREEK T,Reach-1         , 3
Up Type= 0
Dn Type= 3
Dn Slope=0.005
Boundary for River Rch & Prof#=MULBERRY CREEK T,Reach-1         , 4
Up Type= 0
Dn Type= 3
Dn Slope=0.005
Boundary for River Rch & Prof#=MULBERRY CREEK T,Reach-1         , 5
Up Type= 0
Dn Type= 3
Dn Slope=0.005
Boundary for River Rch & Prof#=MULBERRY CREEK T,Reach-1         , 6
Up Type= 0
Dn Type= 3
Dn Slope=0.005
Boundary for River Rch & Prof#=MULBERRY CREEK T,Reach-1         , 7
Up Type= 0
Dn Type= 3
Dn Slope=0.005
DSS Import GetInterval= 0
DSS Import GetPeak= 0
DSS Import FillOption= 0

--- MULBERRY CREEK TRIBUTARY 4.g01 (geometry) ---

Geom Title=Existing Conditions
Program Version=4.10

River Reach=MULBERRY CREEK T,Reach-1
Reach XY= 30
        1568055.        6869588.       1567810.3      6871440.67
      1568644.53      6871978.18       1568660.4      6872690.43
      1569260.38      6873532.83      1569844.52       6873778.2
      1570527.88      6875061.52      1571458.42       6875145.8
      1571844.83      6875528.32      1571958.51      6876329.52
      1572851.45      6877389.47       1573008.5      6878829.54
      1573881.94      6879164.15      1574113.04      6879944.33
      1574951.53       6880739.5      1574855.11      6884217.89
       1574504.7      6885813.12      1574952.95      6886193.84
      1575158.47       6888036.5      1575602.96      6888343.86
      1575255.49      6888948.49      1575358.52      6889636.54
      1576129.53      6889960.86      1576260.45      6890740.47
      1576895.87      6891181.26      1576731.58      6892165.57
       1577257.3      6891993.83       1578170.6       6893037.6
       1579203.6        6892641.        1579155.        6893238.

Type RM Length L Ch R = 1 ,35439   ,339,339,339
BEGIN DESCRIPTION:
MULBERRY CREEK TRIBUTARY 4 53.0
END DESCRIPTION:
XS GIS Cut Line= 3
      1567440.72       6869279.6      1568085.61      6869657.98
      1568655.02        6869688.
#Sta/Elev= 30
  4252.3 1738.95  4326.8 1736.95  4524.8 1734.31  4588.5 1733.71  4597.1 1733.08
  4628.3 1733.55  4744.2 1732.78  4767.2 1731.79    4779 1730.49  4797.3 1731.41
  4810.2 1730.31  4837.4 1729.66  4847.3 1728.33  4883.4 1726.99  4970.4 1727.17
  4976.2 1726.54  5009.4 1726.44  5027.4 1725.65  5027.7 1725.15  5031.2 1725.15
  5031.4 1725.65  5039.4 1727.13  5049.5 1727.77  5059.5 1729.83  5070.8 1729.19
  5284.6 1733.53  5319.8 1734.22  5402.4 1734.27  5530.1 1735.84  5570.2 1737.37
#Mann= 9 ,-1 , 0
  4252.3    .035       0  4524.8     .07       0  4588.5    .035       0
  4797.3     .07       0  5027.4     .07       0  5031.4     .07       0
  5070.8    .035       0  5284.6     .07       0  5402.4    .035       0
Bank Sta=5027.4,5031.4
XS Rating Curve= 0 ,0
Exp/Cntr=0.3,0.1

Type RM Length L Ch R = 1 ,35100   ,447,447,447
BEGIN DESCRIPTION:
MULBERRY CREEK TRIBUTARY 4 52.0
END DESCRIPTION:
XS GIS Cut Line= 3
      1567254.96      6869437.97      1567944.46      6869947.78
      1568786.25      6869974.04
#Sta/Elev= 30
  4142.5 1738.46  4306.4 1733.61  4364.1 1732.71  4492.2 1730.53  4536.1 1730.77
  4615.1  1729.8  4636.3 1730.47  4671.7 1729.19  4717.3 1728.76  4801.2 1727.19
  4828.3 1727.56  4880.4 1725.71  4907.6 1725.73  4928.5 1723.99    4987 1723.99
  4993.2 1723.42  4995.2 1722.42  4995.5 1721.92  4999.2 1722.42  5002.8 1722.42
  5010.5    1724  5063.3 1724.55  5140.6 1725.73  5200.6 1728.16  5300.7 1728.52
  5350.7 1730.15  5370.7  1730.2  5380.7 1729.43  5635.2 1733.65  5842.2 1739.28
#Mann= 8 ,-1 , 0
  4142.5    .035       0  4364.1     .07       0  4717.3    .045       0
  4880.4     .07       0  4995.2     .07       0  4999.2     .07       0
  5063.3    .035       0  5635.2     .07       0
Bank Sta=4995.2,4999.2
XS Rating Curve= 0 ,0
Exp/Cntr=0.3,0.1

Type RM Length L Ch R = 1 ,34653   ,447,447,447
BEGIN DESCRIPTION:
MULBERRY CREEK TRIBUTARY 4 51.0
END DESCRIPTION:
XS GIS Cut Line= 3
      1567055.02      6869638.01        1567905.        6870343.
      1568771.64      6870169.66
#Sta/Elev= 30
  3895.7 1736.26  4051.3 1733.33  4293.5  1728.2  4339.2 1728.27  4428.4 1726.52
  4542.3 1726.68  4577.4 1725.37  4669.9 1724.69  4776.7  1725.1  4805.1 1723.37
  4873.8 1723.11  4953.8 1721.45  4968.1 1720.13  5028.6 1719.66  5028.8 1719.16
  5032.6 1719.66  5048.4  1721.4  5071.4 1721.84  5095.5  1721.1  5265.1 1723.59
  5295.7 1725.27  5410.5 1725.91  5448.7 1727.71  5563.4 1728.47  5609.8 1729.59
  5660.3 1730.99  5665.4 1730.51  5683.3 1732.42  5753.6 1733.92  5883.8 1738.26
#Mann= 9 ,-1 , 0
  3895.7    .035       0  4051.3     .07       0  4339.2    .045       0
  4873.8     .07       0  5028.6     .07       0  5032.6     .07       0
  5095.5    .035       0  5609.8     .07       0  5753.6     .16       0
Bank Sta=5028.6,5032.6
XS Rating Curve= 0 ,0
Exp/Cntr=0.3,0.1

Type RM Length L Ch R = 1 ,34206   ,451,451,451
BEGIN DESCRIPTION:
MULBERRY CREEK TRIBUTARY 4 50.0
END DESCRIPTION:
XS GIS Cut Line= 3
      1567103.04      6870004.42      1567805.23       6870758.1
      1568851.54      6870421.57
#Sta/Elev= 30
  3969.9 1731.64  4143.6  1729.4  4165.1    1728  4200.2 1728.36  4230.1 1726.88
  4277.9 1726.52  4327.7 1724.55  4391.3 1725.37  4405.4 1723.57  4433.8 1722.84
  4497.3 1723.37  4561.3 1721.33    4660 1721.72  4695.6 1720.12  4808.5 1720.11
  4872.5 1717.79  4919.6 1717.81  5019.3 1715.91  5019.6 1715.41  5023.3 1715.91
  5060.9 1717.04  5220.4 1718.85  5325.4 1720.84  5356.9 1722.35  5625.1 1724.78
  5732.5 1723.75  5767.4 1725.31  5840.1 1728.32  5913.6 1729.59  6099.1 1735.81
#Mann= 8 ,-1 , 0
  3969.9     .07       0  4230.1    .045       0  4919.6     .07       0
  5019.3     .07       0  5023.3     .07       0  5060.9    .035       0
  5625.1     .07       0  5767.4     .16       0
Bank Sta=5019.3,5023.3
XS Rating Curve= 0 ,0
Exp/Cntr=0.3,0.1

Type RM Length L Ch R = 1 ,33755   ,624,624,624
BEGIN DESCRIPTION:
MULBERRY CREEK TRIBUTARY 4 49.0
END DESCRIPTION:
XS GIS Cut Line= 3
      1566997.75      6871071.46      1567804.51      6871148.17
      1568984.95      6870507.91
#Sta/Elev= 30
  4189.6 1718.06  4277.2 1717.79  4327.5  1718.6  4407.8 1717.14  4679.1 1716.54
  4749.4 1717.11  4789.5 1715.67  4887.8 1714.58  4990.5 1714.18  5003.1  1713.6
  5006.5  1712.4  5006.8  1711.9  5010.5  1712.4  5030.4 1714.05  5077.7  1714.1
  5296.3 1716.06  5308.9 1716.96  5325.1 1716.41  5353.2 1717.95    5376  1718.2
  5428.7 1717.31  5481.4 1717.46  5710.2 1719.26  5796.9 1720.07  5842.4 1722.21
  5908.9  1723.4  6225.4 1731.92  6289.1 1734.65  6312.9 1735.44  6342.9 1737.95
#Mann= 8 ,-1 , 0
  4189.6    .045       0  4887.8     .07       0  5006.5     .07       0
  5010.5     .07       0  5077.7    .035       0  5481.4     .07       0
  5710.2     .16       0  6289.1     .07       0
Bank Sta=5006.5,5010.5
XS Rating Curve= 0 ,0
Exp/Cntr=0.3,0.1

Type RM Length L Ch R = 1 ,33131   ,650,650,650
BEGIN DESCRIPTION:
MULBERRY CREEK TRIBUTARY 4 48.0
END DESCRIPTION:
XS GIS Cut Line= 3
      1567304.41      6871865.45        1568005.        6871638.
      1568904.99      6870888.01
#Sta/Elev= 30
  4258.8 1714.09  4469.7 1714.36  4521.4 1713.03  4723.7 1713.09  4774.6 1711.75
  4921.8 1711.38  4974.5 1710.08  4992.8 1709.28  5080.6 1709.88  5099.5 1708.28
  5099.7 1707.78  5103.5 1708.28  5115.8 1710.43  5130.1 1711.03  5225.3  1710.6
  5329.6 1710.26  5364.4 1711.34  5393.1 1710.34  5529.2 1711.94  5670.3 1713.11
  5946.3 1719.72  5989.2 1719.71  6105.3 1721.95  6131.1 1722.91  6138.9  1724.8
  6145.4 1724.25  6153.3 1727.41  6159.8 1726.36  6163.7 1727.84  6166.9 1727.84
#Mann= 8 ,-1 , 0
  4258.8    .045       0  4974.5     .07       0  5099.5     .07       0
  5103.5     .07       0  5225.3    .035       0  5329.6     .07       0
  5529.2     .16       0  6105.3     .07       0
#XS Ineff= 2 , 0
       0                  5364.4       0 1711.34
Permanent Ineff=
       F       F
Bank Sta=5099.5,5103.5
XS Rating Curve= 0 ,0
Exp/Cntr=0.3,0.1

Type RM Length L Ch R = 1 ,32481   ,247,247,247
BEGIN DESCRIPTION:
MULBERRY CREEK TRIBUTARY 4 47.0
END DESCRIPTION:
XS GIS Cut Line= 3
      1567464.14      6872167.53      1568462.77       6871844.4
        1568855.        6871238.
#Sta/Elev= 30
  3950.4 1714.47  4094.1 1713.85  4126.1 1714.39  4163.4  1713.1  4277.1 1712.86
  4318.2 1711.39  4413.8  1711.5  4456.7 1710.13    4666  1709.2  4712.8 1710.39
  4718.6 1709.31  4739.5 1708.52  4801.9 1708.78  4936.8 1706.97  4991.8  1705.3
  4996.5 1704.21  4996.8 1703.71  5000.3 1703.71  5000.5 1704.21  5029.3 1705.83
  5351.5 1710.01  5397.3 1711.08  5439.6 1711.06  5475.8 1712.99    5491 1712.46
  5512.1 1712.97  5555.5 1715.53    5615 1717.89  5642.1 1717.98  5722.2 1720.09
#Mann= 6 ,-1 , 0
  3950.4    .045       0  4801.9     .07       0  4996.5     .07       0
  5000.5     .07       0  5029.3     .16       0  5351.5     .07       0
Bank Sta=4996.5,5000.5
XS Rating Curve= 0 ,0
Exp/Cntr=0.3,0.1

Type RM Length L Ch R = 1 ,32234   ,465,465,465
BEGIN DESCRIPTION:
MULBERRY CREEK TRIBUTARY 4 46.0
END DESCRIPTION:
XS GIS Cut Line= 3
      1567754.95      6872388.02        1568655.        6871988.
      1569005.02      6871387.96
#Sta/Elev= 30
  4018.9  1714.5    4038 1714.43  4056.6 1714.71  4079.8 1712.81  4129.9 1712.67
  4161.2 1713.01    4207 1711.28  4270.6 1711.69  4314.4 1709.54  4412.9  1709.8
  4434.8 1708.29  4531.6 1707.06  4806.9 1705.92  4867.7 1704.45  4919.7 1705.12
    4943 1703.73  4947.1    1701  4947.4  1700.5  4951.1    1701  4960.1 1703.06
  4971.7 1703.95  4989.5 1703.42  5165.9  1706.8  5412.8 1709.45  5478.5  1712.6
  5487.2 1711.23    5493 1712.56  5514.5 1711.56  5545.9  1714.6  5698.5 1719.24
#Mann= 6 ,-1 , 0
  4018.9    .045       0    4038     .07       0  4129.9    .045       0
  4531.6     .07       0  4947.1     .07       0  4951.1     .07       0
Bank Sta=4947.1,4951.1
XS Rating Curve= 0 ,0
Exp/Cntr=0.3,0.1

Type RM Length L Ch R = 1 ,31769   ,519,519,519
BEGIN DESCRIPTION:
MULBERRY CREEK TRIBUTARY 4 45.0
END DESCRIPTION:
XS GIS Cut Line= 3
      1568055.01        6872488.        1568705.        6872438.
      1569305.01        6872338.
#Sta/Elev= 30
    4348 1711.65  4378.1    1710    4411 1709.51  4508.5 1708.12  4548.6 1707.19
  4578.7 1705.79  4658.9 1704.87  4789.3 1702.08  4819.4  1702.3  4849.5 1701.25
  4869.5 1701.64  4899.6 1700.92  4959.8  1701.2  4995.4 1700.42  4995.7 1699.92
  4999.2 1699.92  4999.4 1700.42  5032.9  1701.4  5121.6 1701.28  5233.1 1702.21
  5304.1 1704.26  5331.9 1703.77  5354.7 1705.21  5405.4  1705.1    5446 1706.98
  5478.7 1707.05  5496.7 1707.29  5537.2 1709.16  5580.3 1709.57  5608.2 1710.82
#Mann= 5 ,-1 , 0
    4348    .045       0    4411     .07       0  4995.4     .07       0
  4999.4     .07       0  5478.7    .035       0
Bank Sta=4995.4,4999.4
XS Rating Curve= 0 ,0
Exp/Cntr=0.3,0.1

Type RM Length L Ch R = 1 ,31250   ,434,434,434
BEGIN DESCRIPTION:
MULBERRY CREEK TRIBUTARY 4 44.0
END DESCRIPTION:
XS GIS Cut Line= 3
      1567703.03      6872646.08      1568834.97      6872868.08
      1569477.31      6872625.27
#Sta/Elev= 30
  3846.5 1713.22  3934.8 1711.81  4103.3 1710.71  4154.2 1711.54    4192 1709.83
  4254.6 1709.42  4439.6 1706.74  4660.2 1700.56  4755.5 1699.15  4938.9 1697.79
  4989.8 1698.42  5125.2 1697.78  5178.2 1697.02  5178.5 1696.52  5182.2 1697.02
  5203.2 1698.43  5215.8 1700.33  5256.6 1700.17  5288.7 1700.96  5310.1 1702.69
  5325.8 1702.53  5331.4 1703.27  5342.1 1702.62  5354.5 1703.33  5459.7 1707.95
  5481.1 1709.53  5502.5 1709.95    5521 1711.74  5604.4 1713.63  5686.7 1713.89
#Mann= 6 ,-1 , 0
  3846.5    .045       0  4254.6     .07       0  5178.2     .07       0
  5182.2     .07       0  5354.5    .035       0  5604.4     .07       0
Bank Sta=5178.2,5182.2
XS Rating Curve= 0 ,0
Exp/Cntr=0.3,0.1

Type RM Length L Ch R = 1 ,30816   ,290,290,290
BEGIN DESCRIPTION:
Mapping XS ccfceae5
END DESCRIPTION:
XS GIS Cut Line= 4
      1567824.57      6872899.56      1568935.68      6873107.89
      1569324.57      6873135.67       1569508.4       6872802.7
#Sta/Elev= 30
  3718.8 1710.79  3848.9 1710.31  3965.9 1709.14  4334.6 1703.06  4367.9 1701.57
  4493.5 1699.74  4771.9 1697.04  4831.2 1696.58    5009 1694.56  5062.7 1695.91
  5077.2 1692.99  5077.4 1692.49  5081.2 1692.99  5089.2 1693.07  5109.3 1696.49
  5159.4 1696.24  5261.7 1698.77  5295.5  1701.5  5333.4 1700.56  5349.4 1703.53
  5362.1 1708.23  5376.9 1706.39    5385 1702.55    5393 1700.48  5412.3 1702.79
  5458.3 1708.79  5523.6 1709.38  5561.4 1711.71  5590.6  1710.6  5619.5 1711.84
#Mann= 11 ,-1 , 0
  3718.8     .07       0  3848.9    .035       0  3965.9     .07       0
  4367.9    .035       0  4493.5     .07       0  4771.9    .035       0
  4831.2     .07       0  5077.2     .07       0  5081.2     .07       0
  5261.7    .035       0  5412.3     .07       0
Bank Sta=5077.2,5081.2
XS Rating Curve= 0 ,0
Exp/Cntr=0.3,0.1

Type RM Length L Ch R = 1 ,30526   ,487,487,487
BEGIN DESCRIPTION:
Mapping XS f9d4fea2
END DESCRIPTION:
XS GIS Cut Line= 4
      1567994.03      6873839.14       1569233.6      6873328.73
      1569504.43      6873158.59      1569549.49      6872822.37
#Sta/Elev= 30
  3650.2 1707.36  4094.6 1701.83  4256.9  1701.1  4295.7 1699.84    4746 1694.81
  4994.5 1694.35  5005.8 1694.31  5027.8 1694.37  5057.6 1696.86  5072.9 1695.12
  5078.8 1692.66  5086.9 1691.72  5128.6 1691.71  5128.9 1691.21  5132.6 1691.71
  5181.3 1692.45  5188.4 1693.05  5194.3 1695.39  5209.6 1697.34  5299.2 1698.72
  5321.3 1702.22  5341.4 1701.75  5359.6    1703  5381.8 1702.36    5402  1706.5
  5442.3 1706.35  5482.7 1708.83  5553.3 1708.78  5613.9 1711.43  5649.8  1710.5
#Mann= 5 ,-1 , 0
  3650.2     .07       0  5128.6     .07       0  5132.6     .07       0
  5299.2    .035       0  5359.6     .07       0
#XS Ineff= 2 , 0
       0                  5057.6       0 1696.86
Permanent Ineff=
       F       F
Bank Sta=4994.5,5005.8
XS Rating Curve= 0 ,0
Exp/Cntr=0.3,0.1

Type RM Length L Ch R = 1 ,30039   ,189,189,189
BEGIN DESCRIPTION:
Mapping XS 0580722c
END DESCRIPTION:
XS GIS Cut Line= 5
      1568455.85      6874568.27       1569358.6      6873585.67
      1569487.07      6873488.45      1569723.18      6873321.78
      1569653.73      6872974.52
#Sta/Elev= 30
  3502.6 1705.45  3757.1 1702.85  3771.3 1701.22  3785.5 1702.06  3806.4 1700.75
  3948.2 1700.04  3983.4 1698.52  4040.1 1698.57    4394 1694.11  4945.6 1692.99
    4998 1692.88  5004.6 1691.97  5010.7 1692.42  5019.4 1690.99  5044.4 1690.66
  5044.6 1690.16  5048.4 1690.66  5055.1 1692.65    5076 1694.19  5082.1 1693.49
  5090.8  1694.8  5096.9 1693.73  5162.2 1696.05  5355.7 1698.16  5443.9 1700.93
  5464.3 1702.67  5494.9 1701.91  5503.6 1703.47  5529.3 1703.38  5641.2  1705.7
#Mann= 5 ,-1 , 0
  3502.6     .07       0  4945.6    .035       0  5044.4    .035       0
  5048.4    .035       0  5529.3     .07       0
Bank Sta=5044.4,5048.4
XS Rating Curve= 0 ,0
Exp/Cntr=0.3,0.1

Type RM Length L Ch R = 1 ,29850   ,515,515,515
BEGIN DESCRIPTION:
Mapping XS 4c56f905
END DESCRIPTION:
XS GIS Cut Line= 5
      1568553.02      6874745.42      1568799.57      6874439.84
      1569643.32      6873575.25      1569914.15        6873419.
      1569703.23      6873021.36
#Sta/Elev= 30
    3400  1705.1  3619.8 1701.99  3733.4 1702.45  3790.6 1699.91  3910.9 1697.85
  4207.9 1695.74  4469.5    1692  4759.4 1690.83  4793.1 1689.54    4816 1689.11
  4837.3 1694.33  4851.5 1692.02  4964.6 1691.26  4990.9 1688.72  4991.2 1688.22
  4994.9 1688.72  5146.1 1693.27  5316.8 1692.61  5365.2 1694.26  5393.8 1696.97
  5425.5  1696.3    5439 1697.67  5457.5 1697.86  5579.4  1700.4  5595.8 1701.82
  5631.5 1701.06  5654.1 1702.87  5722.4 1703.14  5749.7 1703.96  5763.5 1705.45
#Mann= 6 ,-1 , 0
    3400    .035       0  4793.1     .07       0  4990.9     .07       0
  4994.9     .07       0  5457.5    .035       0  5722.4     .07       0
#XS Ineff= 2 , 0
       0  4837.3 1694.33               0
Permanent Ineff=
       F       F
Bank Sta=4990.9,4994.9
XS Rating Curve= 0 ,0
Exp/Cntr=0.3,0.1

Type RM Length L Ch R = 1 ,29335   ,630,630,630
BEGIN DESCRIPTION:
MULBERRY CREEK TRIBUTARY 4 39.0
END DESCRIPTION:
XS GIS Cut Line= 3
      1568822.83      6874981.16       1569868.2      6874001.73
      1571013.78      6873314.51
#Sta/Elev= 30
  3567.5 1702.08    4165 1695.12  4403.3 1693.81  4766.8 1691.79  4979.3 1688.73
  5153.4 1689.51  5166.9 1687.97  5167.2 1687.47  5170.9 1687.97  5182.7 1689.19
  5334.5 1690.24  5423.6 1689.83  5684.3 1692.92  5707.6 1690.12  5730.7 1691.88
  5736.5 1691.29  5742.6 1693.28  5769.9 1694.47  5800.9 1693.63  5887.3 1694.52
  5892.1 1694.58  6022.2 1695.61    6087 1697.11  6157.8 1699.52  6187.4 1701.05
  6209.1    1701  6232.4 1702.64  6261.3 1702.85  6290.7 1705.25  6335.9  1705.5
#Mann= 11 ,-1 , 0
  3567.5     .07       0    4165    .035       0  4403.3    .045       0
  5166.9    .045       0  5170.9    .045       0  5182.7     .07       0
  5769.9    .035       0  5887.3     .07       0  5892.1    .035       0
    6087     .07       0  6157.8    .035       0
Bank Sta=5166.9,5170.9
XS Rating Curve= 0 ,0
Exp/Cntr=0.3,0.1

Type RM Length L Ch R = 1 ,28705   ,428,428,428
BEGIN DESCRIPTION:
MULBERRY CREEK TRIBUTARY 4 38.0
END DESCRIPTION:
XS GIS Cut Line= 3
        1569455.        6875138.      1570278.39      6874411.31
      1571350.28       6873498.8
#Sta/Elev= 30
  3901.8 1696.05    4127  1693.6  4256.1 1693.69  4262.8 1692.85  4432.5 1691.94
  4702.1 1688.97  4723.7 1689.51    4830 1687.16  4907.8 1687.15  4998.7 1686.39
  5141.4 1688.05  5155.7 1687.11  5163.4 1687.73    5170 1685.54  5177.7 1686.36
  5182.2 1684.94  5182.5 1684.44  5186.2 1684.94  5227.1 1688.03  5255.6 1686.87
  5358.1 1687.65  5638.9 1689.34  5746.5 1691.32  5826.8 1693.25    5857  1694.1
  6203.4 1701.91  6227.5 1701.64  6256.1 1703.63  6312.8 1704.14  6407.7 1705.91
#Mann= 12 ,-1 , 0
  3901.8     .07       0    4127    .035       0  4432.5    .045       0
  4907.8     .07       0  5182.2     .07       0  5186.2     .07       0
  5358.1    .035       0  5746.5     .07       0  5826.8    .035       0
    5857     .07       0  6203.4    .035       0  6312.8     .07       0
Bank Sta=5182.2,5186.2
XS Rating Curve= 0 ,0
Exp/Cntr=0.3,0.1

Type RM Length L Ch R = 1 ,28277   ,561,561,561
BEGIN DESCRIPTION:
MULBERRY CREEK TRIBUTARY 4 37.0
END DESCRIPTION:
XS GIS Cut Line= 3
      1569485.18      6875659.95      1570455.45      6874772.81
      1571362.53      6873671.73
#Sta/Elev= 30
  3685.3 1699.54  4033.5 1692.96  4394.2 1690.45  4599.6 1688.85  4656.4 1689.61
  4727.3 1687.18  5022.3 1683.78  5022.5 1683.28  5026.3 1683.78  5069.6 1685.11
  5264.7 1686.12  5322.7 1685.59  5351.4  1683.9  5380.1 1685.62  5464.6 1685.38
  5586.3 1686.66    5728 1688.59  5742.3 1689.44  5763.1 1694.05  5783.9 1696.35
  5791.8 1696.36  5798.3 1693.31  5806.2 1692.83  5812.6 1690.81  5820.5 1691.24
    5827 1688.79  5841.3 1688.32  6061.5 1696.74  6125.4 1696.88  6426.6 1702.23
#Mann= 8 ,-1 , 0
  3685.3     .07       0  4394.2    .035       0  5022.3    .035       0
  5026.3    .035       0  5069.6    .045       0  5264.7     .07       0
  5464.6    .035       0  5586.3     .07       0
#XS Ineff= 2 , 0
       0                  5279.7       0 1686.66
Permanent Ineff=
       F       F
Bank Sta=5022.3,5026.3
XS Rating Curve= 0 ,0
Exp/Cntr=0.3,0.1

Type RM Length L Ch R = 1 ,27716   ,907,907,907
BEGIN DESCRIPTION:
MULBERRY CREEK TRIBUTARY 4 36.0
END DESCRIPTION:
XS GIS Cut Line= 3
      1569648.33      6876032.56        1570705.        6875238.
      1571676.14      6873548.84
#Sta/Elev= 30
  3674.1  1703.5  3895.5 1696.31  4082.8 1691.97  4189.9 1691.37  4272.3 1689.57
  4382.8 1689.01  4389.1  1686.8  4403.7 1687.03  4424.5 1685.52  4439.1  1687.3
  4459.9 1691.98  4468.2 1691.79  4495.7 1687.28  4574.8 1686.62    4993 1682.31
  5245.6 1682.96  5329.8 1682.09  5330.1 1681.59  5333.8 1682.09  5406.6 1683.41
  5642.1 1683.14  5765.9 1686.01  5830.6 1690.01  5926.9 1691.83  6211.6 1691.98
  6493.3 1694.92  6560.9 1696.14  6808.6 1699.86  6919.3 1704.73  6944.6 1705.52
#Mann= 10 ,-1 , 0
  3674.1     .07       0  4189.9    .045       0  4272.3     .07       0
  4574.8    .045       0  5329.8    .045       0  5333.8    .045       0
  6493.3    .035       0  6560.9     .07       0  6808.6    .035       0
  6919.3     .07       0
Bank Sta=5329.8,5333.8
XS Rating Curve= 0 ,0
Exp/Cntr=0.3,0.1

Type RM Length L Ch R = 1 ,26809   ,494,494,494
BEGIN DESCRIPTION:
MULBERRY CREEK TRIBUTARY 4 35.0
END DESCRIPTION:
XS GIS Cut Line= 3
      1569905.02      6876437.99        1571505.        6875188.
        1571805.        6873988.
#Sta/Elev= 30
  2969.2 1701.15  3019.8 1699.05  3056.1 1698.66  3517.3 1689.59  4259.2 1683.93
  4337.5  1682.6  4401.7 1682.33  4451.5  1682.3  4486.8 1683.36    4522 1681.64
  4620.7 1681.14  4855.2 1679.56  4855.5 1679.06  4859.6 1679.06    4860 1679.56
  4956.7    1680  5022.8 1679.79  5182.5 1680.75  5223.8 1681.17  5236.7 1682.07
  5558.8 1684.63  5896.3 1689.68  6053.5 1690.82  6177.2    1694    6185 1694.48
  6205.6 1698.57  6213.3 1701.41  6218.5 1699.84  6226.2  1702.6  6236.5 1702.04
#Mann= 7 ,-1 , 0
  2969.2     .07       0  3056.1    .045       0  4259.2     .07       0
  4620.7    .045       0  4855.2     .07       0    4860    .045       0
  4956.7     .07       0
Bank Sta=4855.2,4860
XS Rating Curve= 0 ,0
Exp/Cntr=0.3,0.1

Type RM Length L Ch R = 1 ,26315   ,420,420,420
BEGIN DESCRIPTION:
MULBERRY CREEK TRIBUTARY 4 34.0
END DESCRIPTION:
XS GIS Cut Line= 3
      1570057.06      6876515.09      1571657.08      6875715.08
      1572828.03      6874653.21
#Sta/Elev= 30
  2948.7 1697.59  3377.5 1689.31  3502.9 1688.22  3679.3 1686.51  3727.4 1686.15
  3839.7 1685.15  3867.1 1685.02  4038.4 1684.14  4241.6 1681.85  4419.3 1680.69
  4624.4 1679.64  4719.2    1678  4889.8 1677.98  4932.4    1676  4995.9 1677.91
    5015 1675.35  5015.4 1674.85    5020 1675.35  5038.5 1677.47  5066.8 1676.64
    5102 1678.09  5144.6 1677.05  5229.7 1678.43  5314.9 1678.05    5510 1680.36
  5590.6  1682.2  5633.2  1684.4  5902.1  1690.6  5930.5 1692.17  6318.3  1698.6
#Mann= 13 ,-1 , 0
  2948.7    .045       0  3502.9     .07       0  3679.3    .045       0
  3727.4     .07       0  3839.7    .045       0  3867.1    .035       0
  4038.4    .045       0  4241.6    .035       0  4419.3    .045       0
  4624.4     .07       0    5015     .07       0    5020     .07       0
    5510    .035       0
Bank Sta=5015,5020
XS Rating Curve= 0 ,0
Exp/Cntr=0.3,0.1

Type RM Length L Ch R = 1 ,25895   ,475,475,475
BEGIN DESCRIPTION:
MULBERRY CREEK TRIBUTARY 4 33.0
END DESCRIPTION:
XS GIS Cut Line= 3
      1570140.51      6876653.22        1571855.        6875888.
      1572920.93       6874773.9
#Sta/Elev= 30
    3127 1695.66  3416.6 1690.54  3698.3 1687.47  4156.2 1683.92  4467.9 1680.38
  4511.7 1679.17    4665  1678.4  4700.6 1679.25    4722 1678.09  4897.3 1677.45
  4999.1 1675.15  4999.6 1674.65  5004.4 1675.15  5068.2 1675.54  5082.3  1676.4
  5103.4 1675.33  5145.9 1675.49  5167.3 1676.79  5188.3 1675.77  5195.6 1676.96
  5202.5 1675.88  5223.9 1676.78  5230.8 1675.73  5287.4 1675.53  5379.2 1677.98
  5421.7 1677.06    5634    1680  5680.3 1682.53  6249.5 1693.33  6546.4 1698.03
#Mann= 7 ,-1 , 0
    3127    .045       0  3698.3    .035       0  4156.2    .045       0
    4722     .07       0  4999.1     .07       0  5004.4     .07       0
  5680.3    .035       0
Bank Sta=4999.1,5004.4
XS Rating Curve= 0 ,0
Exp/Cntr=0.3,0.1

Type RM Length L Ch R = 1 ,25420   ,566,566,566
BEGIN DESCRIPTION:
MULBERRY CREEK TRIBUTARY 4 32.0
END DESCRIPTION:
XS GIS Cut Line= 3
      1570182.24      6876752.16        1571955.        6876338.
      1573005.11      6874913.65
#Sta/Elev= 30
  3171.3 1694.41  3233.2 1693.36  3437.9 1690.97  3523.8 1689.25  3841.8 1686.55
  4399.8 1681.79    4581 1679.09  4611.8 1679.87  4617.6  1678.6  4627.6 1678.27
  4765.9 1675.25  4929.2  1674.3  4994.9 1673.26  5002.6 1671.97  5003.1 1671.47
    5008 1671.97  5049.2 1673.62    5132 1673.96  5133.4    1674  5252.1 1674.79
  5285.8 1674.51  5341.6 1674.38  5522.9 1676.52  5674.4 1678.66  5999.4 1684.08
  6099.7 1684.64  6206.2 1687.18  6358.6 1689.43  6500.7 1692.33  6761.4 1695.75
#Mann= 16 ,-1 , 0
  3171.3    .045       0  3233.2     .07       0  3437.9    .035       0
  3841.8    .045       0  4627.6     .07       0  4929.2    .035       0
  5002.6    .035       0    5008    .035       0    5132     .07       0
  5133.4    .035       0  5252.1     .07       0  5285.8    .035       0
  5522.9     .07       0  5674.4    .035       0  6206.2     .07       0
  6358.6    .035       0
Bank Sta=5002.6,5008
XS Rating Curve= 0 ,0
Exp/Cntr=0.3,0.1

Type RM Length L Ch R = 1 ,24854   ,352,352,352
BEGIN DESCRIPTION:
MULBERRY CREEK TRIBUTARY 4 31.0
END DESCRIPTION:
XS GIS Cut Line= 3
      1570244.73      6876851.12        1572255.        6876763.
      1573479.08      6876408.42
#Sta/Elev= 30
  2987.8 1692.14  3081.6 1690.74  3180.8 1689.66  3378.4 1687.28  3678.7 1686.22
  3893.3 1684.42    4009 1683.32    4227 1680.39  4374.7 1678.38    4485 1676.77
  4710.7 1671.86  4899.9 1671.34  4929.9 1670.52  4936.9 1669.36  4937.4 1668.86
  4942.9 1669.36    4950 1670.41    4970 1671.02    5000 1670.14  5103.4 1672.16
  5173.1 1672.03    5427 1673.06  5812.1 1677.04  5853.7 1679.22  5917.7 1681.16
  5971.9 1682.76    6011 1684.99  6077.9 1687.15  6249.3  1688.7  6274.4 1690.49
#Mann= 15 ,-1 , 0
  2987.8    .035       0  3081.6     .07       0  3180.8    .035       0
  3893.3     .07       0    4009    .035       0    4227     .07       0
  4374.7    .035       0    4485     .07       0  4710.7    .035       0
  4936.9    .035       0  4942.9    .035       0  5173.1     .07       0
    5427    .035       0  5917.7     .07       0    6011    .035       0
Bank Sta=4936.9,4942.9
XS Rating Curve= 0 ,0
Exp/Cntr=0.3,0.1

Type RM Length L Ch R = 1 ,24502   ,949,949,949
BEGIN DESCRIPTION:
Mapping XS 306d8f3e
END DESCRIPTION:
XS GIS Cut Line= 3
      1569622.42      6878021.14      1572405.08      6877062.98
      1573475.25        6876611.
#Sta/Elev= 30
    2057 1691.61  2484.7 1688.54  2848.8 1683.79  2854.1 1684.72  2911.2 1684.63
  3280.6 1680.09    3369 1677.89  3400.2  1676.1  3499.1 1678.68  3743.6 1679.35
  4170.2 1675.36  4477.1 1674.38  4659.1 1671.64  4695.6  1670.2  4752.8  1670.1
  4786.3 1668.15  4786.8 1667.65  4792.4 1668.15  4841.2 1670.24  4883.6 1670.63
  4915.3 1669.02  4978.8 1669.68  5010.8 1668.66  5043.3 1670.09  5338.9 1671.16
    5508 1672.76  5759.8 1677.87  5803.2 1680.72  5950.3 1685.19  6161.7 1686.52
#Mann= 5 ,-1 , 0
    2057    .035       0  4786.3    .035       0  4792.4    .035       0
  5338.9     .07       0    5508    .035       0
Bank Sta=4786.3,4792.4
XS Rating Curve= 0 ,0
Exp/Cntr=0.3,0.1

Type RM Length L Ch R = 1 ,23553   ,555,555,555
BEGIN DESCRIPTION:
MULBERRY CREEK TRIBUTARY 4 30.0
END DESCRIPTION:
XS GIS Cut Line= 3
      1570457.47      6878689.55        1572855.        6877638.
      1573605.03      6877037.98
#Sta/Elev= 30
  2381.9    1698  2450.5 1697.64  2641.7 1692.44  2881.5 1686.46  3123.3 1683.04
  3351.4 1680.69  3589.5 1677.65  3996.2 1668.04  4071.7 1670.06  4287.5  1671.5
  4657.8 1667.85  4743.6 1667.51  4909.9 1666.38  4938.7 1667.46  4987.2 1665.98
  4987.7 1665.48  4994.7 1665.98  4997.2 1667.13  5013.5 1667.41  5234.4 1667.16
  5650.5  1672.3  5690.6 1672.86  5725.9 1676.71  5732.3 1678.46  5761.1 1679.98
  5888.8  1682.8  5938.8 1683.92  5953.2 1687.87  5957.2 1690.63  5960.4 1690.63
#Mann= 11 ,-1 , 0
  2381.9    .035       0  2450.5     .07       0  2641.7    .035       0
  3123.3     .07       0  3351.4    .035       0  4657.8     .07       0
  4743.6    .035       0  4987.2    .035       0  4994.7    .035       0
  5650.5     .07       0  5888.8    .035       0
Bank Sta=4987.2,4994.7
XS Rating Curve= 0 ,0
Exp/Cntr=0.3,0.1

Type RM Length L Ch R = 1 ,22998   ,358,358,358
BEGIN DESCRIPTION:
MULBERRY CREEK TRIBUTARY 4 29.0
END DESCRIPTION:
XS GIS Cut Line= 3
      1571423.07      6879269.11      1572806.71      6878077.25
        1573655.        6877388.
#Sta/Elev= 30
  3173.8 1689.93    3241 1689.27  3395.9 1686.68  3445.3 1683.02  3891.8 1672.54
  4118.9 1669.56  4338.4 1668.23  4452.5 1665.64    4615  1664.7  4682.4 1663.35
  4682.9 1662.85    4690 1663.35  4728.9 1665.09  4757.5 1663.69    4786 1664.74
  4835.4 1664.26  4941.8 1665.88  4958.1 1665.12  4962.6 1664.83  5040.7 1666.06
  5138.4 1666.11  5139.3 1666.14    5282 1665.22  5547.2 1669.71  5609.6 1670.15
  5723.1 1672.87  5826.7 1677.32    5894 1679.17  6010.2 1680.16    6093 1680.57
#Mann= 11 ,-1 , 0
  3173.8     .07       0    3241    .035       0  4682.4    .035       0
    4690    .035       0  4958.1     .07       0  4962.6    .035       0
  5138.4     .07       0  5139.3    .035       0  5547.2     .07       0
  5826.7    .035       0  6010.2     .07       0
Bank Sta=4682.4,4690
XS Rating Curve= 0 ,0
Exp/Cntr=0.3,0.1

Type RM Length L Ch R = 1 ,22640   ,450,450,450
BEGIN DESCRIPTION:
MULBERRY CREEK TRIBUTARY 4 28.0
END DESCRIPTION:
XS GIS Cut Line= 3
      1571754.97      6879288.03        1572955.        6878388.
      1573704.98      6877888.02
#Sta/Elev= 30
    3499 1687.62  3527.2 1684.75  3606.3  1680.3  3920.9 1670.93  3927.2 1671.73
  4070.9  1668.9  4341.8 1666.66    4399    1663  4441.8 1663.27  4456.3 1662.28
  4462.6 1663.38  4491.8 1663.63  4535.5 1662.68  4656.3 1663.82  4777.2 1663.55
  4802.5 1662.13    4803 1661.63  4810.1 1662.13  4835.5 1663.52  4891.8 1663.95
  5078.7 1664.41  5143.3 1663.59  5251.4 1666.33  5258.9 1667.34    5301 1667.65
  5388.1 1672.02  5460.3 1672.89  5475.3    1674  5553.4 1674.16  5900.4 1680.53
#Mann= 3 ,-1 , 0
    3499    .035       0  4802.5    .035       0  4810.1    .035       0
Bank Sta=4802.5,4810.1
XS Rating Curve= 0 ,0
Exp/Cntr=0.3,0.1

Type RM Length L Ch R = 1 ,22190   ,194,194,194
BEGIN DESCRIPTION:
MULBERRY CREEK TRIBUTARY 4 27.0
END DESCRIPTION:
XS GIS Cut Line= 3
      1571804.98      6879388.01        1573005.        6878788.
      1573708.89      6877952.17
#Sta/Elev= 30
  3663.2 1687.12  3716.3 1685.52  3744.3 1684.22    3789 1680.76  3856.1  1678.2
  3962.3 1674.31  4155.2 1668.88  4311.7 1668.07    4566 1662.54  4669.5 1661.54
  4705.8 1662.15  4728.2 1661.66  4755.3  1662.5  4793.8 1662.25  4817.6 1660.89
  4862.3 1662.39  4884.7 1662.33  4901.4 1661.27  4982.5 1662.25  5002.1 1661.12
  5036.8  1660.7  5037.3  1660.2  5044.4  1660.7  5075.7 1662.54  5203.2 1664.26
  5352.7  1669.6  5458.3 1671.37    5644 1674.19  5853.7 1675.51  6097.6 1680.22
#Mann= 7 ,-1 , 0
  3663.2    .035       0  4755.3     .07       0  4793.8    .035       0
  5036.8    .035       0  5044.4    .035       0  5458.3     .07       0
  5853.7    .035       0
Bank Sta=5036.8,5044.4
XS Rating Curve= 0 ,0
Exp/Cntr=0.3,0.1

Type RM Length L Ch R = 1 ,21996   ,651,651,651
BEGIN DESCRIPTION:
MULBERRY CREEK TRIBUTARY 4 26.0
END DESCRIPTION:
XS GIS Cut Line= 3
      1571850.15      6880138.91      1573144.37      6878889.51
      1573730.17      6878029.82
#Sta/Elev= 30
  3201.1  1683.8  3339.5 1682.73  3693.3 1672.03  3707.4 1672.44  3763.8 1671.01
    3807 1670.89  4122.3 1666.78  4145.8 1667.12  4188.2 1666.04  4301.4 1665.33
  4556.1 1661.03  4576.9 1661.51    4587 1661.31  4676.2 1660.85  4824.7 1661.84
  4930.9 1659.58  4937.9  1660.6  4962.3 1658.89  4962.8 1658.39  4969.9 1658.89
  4987.2 1660.65    5037 1661.19  5152.6 1663.29    5200 1664.94  5332.1 1669.16
  5583.5 1673.26  5671.8 1673.68  5836.8 1675.02  5873.8 1675.97  6040.3 1679.35
#Mann= 11 ,-1 , 0
  3201.1    .035       0    3807     .07       0  4122.3    .035       0
  4576.9     .07       0    4587    .035       0  4962.3    .035       0
  4969.9    .035       0    5037     .07       0    5200    .035       0
  5671.8     .07       0  5873.8    .035       0
Bank Sta=4962.3,4969.9
XS Rating Curve= 0 ,0
Exp/Cntr=0.3,0.1

Type RM Length L Ch R = 1 ,21345   ,740,740,740
BEGIN DESCRIPTION:
MULBERRY CREEK TRIBUTARY 4 25.0
END DESCRIPTION:
XS GIS Cut Line= 3
      1572272.08      6880232.61        1573655.        6879038.
      1573756.43      6878123.25
#Sta/Elev= 30
  3177.5 1678.72  3218.6  1677.8    3381 1671.81  3601.4 1667.26  4387.9 1658.19
  4572.4 1659.47    4728 1659.71  4742.3 1658.93  4749.9 1657.29  4756.5 1657.67
  4764.2 1659.81  4783.9 1659.76  4790.4  1659.7  4962.7 1658.84    4977 1658.59
  4979.4 1657.04  4979.9 1656.54  4987.7 1657.04  5007.5 1657.31    5015 1658.66
  5045.2 1659.55  5050.3 1660.58  5055.3 1660.54  5085.4 1665.45  5105.6 1666.65
  5183.6  1667.7  5377.2 1671.14  5812.5 1675.21  5843.2 1675.55  5925.3  1676.5
#Mann= 9 ,-1 , 0
  3177.5    .035       0  4572.4     .07       0  4783.9    .035       0
  4790.4     .07       0  4979.4     .07       0  4987.7     .07       0
  5183.6    .035       0  5812.5     .07       0  5843.2    .035       0
Bank Sta=4979.4,4987.7
XS Rating Curve= 0 ,0
Exp/Cntr=0.3,0.1

Type RM Length L Ch R = 1 ,20605   ,404,404,404
BEGIN DESCRIPTION:
MULBERRY CREEK TRIBUTARY 4 24.0
END DESCRIPTION:
XS GIS Cut Line= 3
      1572355.01        6880288.      1573978.01      6879561.47
      1574584.53      6878555.58
#Sta/Elev= 30
  3221.8 1677.72  3316.1 1675.66  3843.2 1664.96  4222.1 1659.87    4248 1659.63
  4404.2 1658.28    4416 1660.93  4432.9 1661.49  4438.4 1663.88  4470.8 1659.82
  4484.8 1656.11  4492.7 1657.65  4652.6 1656.24  4832.4 1657.23  4924.2 1656.56
  4947.3 1655.95  4948.6  1654.9  4949.1  1654.4  4957.1  1654.9  4963.6 1654.93
  5038.7 1657.26  5195.8 1657.85  5218.5 1658.42  5239.8 1661.16  5283.9 1662.75
  5295.6 1663.06  5398.9 1665.83  5833.4 1671.72  5992.3 1672.77  6174.6  1674.8
#Mann= 15 ,-1 , 0
  3221.8    .035       0  3316.1     .07       0  3843.2    .035       0
  4222.1     .07       0    4248    .035       0  4948.6     .07       0
  4957.1    .035       0  4963.6     .07       0  5038.7    .035       0
  5195.8     .07       0  5283.9    .035       0  5295.6     .07       0
  5398.9    .035       0  5833.4     .07       0  5992.3    .035       0
Bank Sta=4948.6,4957.1
XS Rating Curve= 0 ,0
Exp/Cntr=0.3,0.1

Type RM Length L Ch R = 1 ,20201   ,420,420,420
BEGIN DESCRIPTION:
MULBERRY CREEK TRIBUTARY 4 23.0
END DESCRIPTION:
XS GIS Cut Line= 3
      1572654.99        6880338.      1574075.22      6879857.84
      1574693.93      6878628.46
#Sta/Elev= 30
  3500.8 1672.91  3592.2 1671.79  3881.9 1667.43  4037.2  1665.4  4342.2 1660.69
  4936.4  1655.8  4992.9 1653.22  4993.4 1652.72  5001.6 1653.22  5013.6  1654.7
  5044.6 1656.05    5075 1655.99  5119.6 1654.09  5193.1 1655.96    5250  1655.8
  5383.5  1655.7  5491.6 1657.26  5675.2 1660.78    5816 1664.17  5967.7 1663.19
  6015.2 1663.84  6034.6 1663.66  6073.7 1666.33  6079.3 1665.86    6096 1669.33
  6101.6 1667.97  6118.3 1670.71  6140.6 1672.12  6335.7 1675.62  6376.3 1675.89
#Mann= 15 ,-1 , 0
  3500.8    .035       0  3592.2     .07       0  3881.9    .035       0
  4037.2     .07       0  4342.2    .035       0  4992.9    .035       0
  5001.6    .035       0  5193.1     .07       0    5250    .035       0
  5383.5     .07       0  5491.6    .035       0  5675.2     .07       0
    5816    .035       0  6015.2     .07       0  6335.7    .035       0
Bank Sta=4992.9,5001.6
XS Rating Curve= 0 ,0
Exp/Cntr=0.3,0.1

Type RM Length L Ch R = 1 ,19781   ,704,704,704
BEGIN DESCRIPTION:
MULBERRY CREEK TRIBUTARY 4 21.0
END DESCRIPTION:
XS GIS Cut Line= 3
      1572813.73      6880503.46      1574352.81      6880143.99
      1575000.62      6878890.04
#Sta/Elev= 30
  3419.5  1671.7  3531.2 1670.82  3977.3 1665.34    4479  1659.4  4541.4 1658.61
  4632.6 1656.86  4746.1 1655.79  4765.7  1655.6  4940.6 1654.66  4963.3    1653
  4967.1 1651.37  4967.6 1650.87  4975.8 1651.37  4981.7  1652.7    4992  1653.6
  5019.6 1654.85  5163.4 1653.69  5191.2 1652.57  5207.7 1653.24  5220.6 1652.25
  5265.6  1653.8  5296.3 1652.73  5355.7 1653.74  5445.7 1653.47  5642.3 1655.44
  5977.3 1660.62  6053.5  1664.5  6082.4 1667.76  6303.9 1670.78  6411.4 1673.14
#Mann= 10 ,-1 , 0
  3419.5    .035       0  3531.2     .07       0  3977.3    .035       0
    4479     .07       0  4541.4    .035       0  4746.1     .07       0
  4765.7    .035       0  4967.1    .035       0  4975.8    .035       0
  5642.3     .07       0
Bank Sta=4967.1,4975.8
XS Rating Curve= 0 ,0
Exp/Cntr=0.3,0.1

Type RM Length L Ch R = 1 ,19077   ,467,467,467
BEGIN DESCRIPTION:
MULBERRY CREEK TRIBUTARY 4 20.0
END DESCRIPTION:
XS GIS Cut Line= 3
      1573099.17      6880526.18        1574755.        6880538.
        1575055.      6879338.01
#Sta/Elev= 30
  3335.9 1668.71  3398.8 1667.98  3781.7 1664.53  3941.7 1662.06  4341.8 1658.88
  4371.8 1659.53  4561.8 1659.21  4875.2 1655.55  4951.8 1654.24  4989.3 1651.82
    5051 1652.13  5069.8 1651.02  5070.3 1650.52  5078.6 1651.02  5105.2 1652.69
  5124.1 1652.71  5221.1 1651.86  5257.2 1652.36  5303.6 1651.15  5344.8 1652.97
  5503.6 1652.93    5659 1653.18  5847.3 1654.02  5867.9 1654.42  5880.8  1655.9
  5909.2 1655.42  5963.3 1657.43  6040.6 1661.73  6074.1 1665.85  6228.7 1667.21
#Mann= 8 ,-1 , 0
  3335.9     .07       0  3398.8    .035       0  4875.2     .07       0
  5069.8     .07       0  5078.6     .07       0  5124.1    .035       0
  5503.6     .07       0    5659    .035       0
Bank Sta=5069.8,5078.6
XS Rating Curve= 0 ,0
Exp/Cntr=0.3,0.1

Type RM Length L Ch R = 1 ,18610   ,467,467,467
BEGIN DESCRIPTION:
MULBERRY CREEK TRIBUTARY 4 19.0
END DESCRIPTION:
XS GIS Cut Line= 3
      1573174.85      6880625.95        1574905.        6880888.
      1577465.41       6880732.6
#Sta/Elev= 30
  3245.4 1667.74  4125.5  1660.2  4590.7 1658.75  4782.9 1656.24  4904.1 1653.06
  4997.8 1650.31  5035.4 1650.38  5051.6 1650.05  5079.1 1651.27  5196.3 1651.12
  5240.9 1651.61  5345.9 1651.81    5376 1650.37  5409.5 1651.48  5556.6 1651.05
  5737.1 1649.75  5812.3 1648.58  5812.8 1648.08  5821.2 1648.58  5856.9 1649.99
  6007.1 1650.39  6245.8 1653.89    6639 1658.97  6678.4 1658.15  6748.5 1659.52
  6798.6 1663.15  6827.2 1663.11  6982.7 1663.83  7557.6 1666.69  7560.4 1666.69
#Mann= 14 ,-1 , 0
  3245.4    .035       0  4904.1     .07       0  5051.6    .035       0
  5196.3     .07       0  5240.9    .035       0  5556.6     .07       0
  5737.1    .035       0  5812.3     .07       0  5821.2    .035       0
  6245.8     .07       0    6639    .035       0  6827.2     .07       0
  6982.7    .035       0  7557.6     .07       0
#XS Ineff= 2 , 0
       0                  5335.9       0    1654
Permanent Ineff=
       F       F
Bank Sta=4997.8,5035.4
XS Rating Curve= 0 ,0
Exp/Cntr=0.3,0.1

Type RM Length L Ch R = 1 ,18143   ,468,468,468
BEGIN DESCRIPTION:
MULBERRY CREEK TRIBUTARY 4 18.0
END DESCRIPTION:
XS GIS Cut Line= 3
      1572868.23      6880892.49        1574955.        6881338.
      1577420.12      6881454.99
#Sta/Elev= 30
  2866.2 1669.38  3034.9 1667.99  3257.3 1666.32  4488.7 1658.44  4930.8 1653.32
  4975.2 1649.24    5010 1651.86    5040 1649.49  5080.1 1649.42  5288.8 1649.39
  5596.2 1648.27  5703.2 1649.11  5785.4 1647.73  5806.5 1647.53    5807 1647.03
  5815.4 1647.53  6091.6 1648.96  6165.8 1648.86  6282.9 1649.75  6631.8 1658.13
  6749.2 1663.56  6791.6 1664.29  7027.2  1666.8  7035.2 1666.83  7187.5 1668.73
  7232.5 1670.44  7262.5 1674.17  7311.5 1675.11  7351.1 1675.59  7467.9  1677.8
#Mann= 19 ,-1 , 0
  2866.2    .035       0  3034.9     .07       0  3257.3    .035       0
  5288.8     .07       0  5596.2    .035       0  5703.2     .07       0
  5785.4    .035       0  5806.5    .035       0  5815.4    .035       0
  6091.6     .07       0  6165.8    .035       0  6282.9     .07       0
  6749.2    .035       0  6791.6    .063       0  7027.2    .094       0
  7035.2    .063       0  7187.5    .094       0  7311.5    .063       0
  7351.1    .094       0
#XS Ineff= 2 , 0
       0                  5700.8       0    1651
Permanent Ineff=
       F       F
Bank Sta=5040,5080.1
XS Rating Curve= 0 ,0
Exp/Cntr=0.3,0.1

Type RM Length L Ch R = 1 ,17675   ,560,560,560
BEGIN DESCRIPTION:
MULBERRY CREEK TRIBUTARY 4 17.0
END DESCRIPTION:
XS GIS Cut Line= 3
      1572764.09      6881559.17        1575005.        6881788.
      1576920.17      6882027.89
#Sta/Elev= 30
  2742.4 1668.54  3306.2 1661.25  3586.4 1662.18    3610 1662.04    4532 1654.51
  4541.9 1654.15  4682.4    1650  4896.2 1647.96  4984.9 1646.79    5005 1646.81
  5260.6  1647.6  5329.5 1647.54  5544.8 1645.42  5545.3 1644.92  5553.7 1645.42
  5762.6 1645.67    5854 1650.94  6194.3 1649.38    6285 1653.39  6321.4 1647.13
    6334 1648.82  6385.7 1649.71  6436.1 1657.78  6456.3 1655.11  6507.5 1656.74
    6563 1663.78  6724.1 1665.35  6785.8 1670.74  6859.4 1674.62  6925.1 1673.23
#Mann= 15 ,-1 , 0
  2742.4    .035       0  3586.4     .07       0    3610    .035       0
    4532     .07       0  4541.9    .035       0  4682.4     .07       0
  4896.2    .035       0  5260.6     .07       0  5329.5    .035       0
  5544.8    .035       0  5553.7    .035       0    5854     .07       0
    6334    .035       0  6507.5    .063       0  6785.8    .094       0
Bank Sta=4984.9,5005
XS Rating Curve= 0 ,0
Exp/Cntr=0.3,0.1

Type RM Length L Ch R = 1 ,17115   ,531,531,531
BEGIN DESCRIPTION:
Mapping XS c03023e0
END DESCRIPTION:
XS GIS Cut Line= 3
      1572804.91      6882022.71      1574883.89      6882278.78
      1576331.76      6882374.15
#Sta/Elev= 30
  2884.1 1667.67    3126 1666.69  3962.3 1654.18  4029.7 1655.54  4234.3 1655.53
  4735.3 1648.38  4834.7 1645.85  4927.1  1644.4  5029.8 1644.64  5210.4 1645.26
  5396.3 1643.12  5396.8 1642.62  5405.3 1643.12  5571.2 1645.06  5691.4 1643.48
  5731.5 1644.86  5831.7 1644.66  6000.6 1646.54  6062.2 1649.62  6072.3 1652.35
  6107.7 1656.93  6112.7  1656.5  6132.4 1658.95  6149.1 1659.32  6200.3 1659.84
  6242.6 1658.25  6320.8 1660.47  6332.8 1660.48  6362.9 1663.09  6429.8 1663.25
#Mann= 11 ,-1 , 0
  2884.1    .035       0  4735.3     .07       0  4834.7    .035       0
  4927.1     .07       0  5029.8    .035       0  5396.3     .07       0
  5405.3    .035       0  6000.6     .07       0  6149.1    .035       0
  6200.3     .07       0  6320.8    .063       0
Bank Sta=5396.3,5405.3
XS Rating Curve= 0 ,0
Exp/Cntr=0.3,0.1

Type RM Length L Ch R = 1 ,16584   ,415,415,415
BEGIN DESCRIPTION:
Mapping XS 44f38353
END DESCRIPTION:
XS GIS Cut Line= 3
      1573134.71       6882647.7      1574927.29      6882743.19
      1576050.68      6882626.08
#Sta/Elev= 30
  3184.8 1659.64  3315.3 1658.95  3455.5 1659.75  3631.2 1657.89  3725.2 1656.25
    3977 1654.66  4167.6 1650.88  4222.9 1649.15  4456.9 1645.34  4577.1 1645.99
  4647.2 1643.59  4707.2 1643.12  4747.3 1644.23  4983.1  1641.6  4983.6  1641.1
  4992.2  1641.6  5096.6 1642.68  5196.7 1642.97  5440.1 1642.73  5482.8 1643.68
  5656.6 1643.94    5746 1645.68  5842.3 1648.69  5882.5 1650.98  5892.6 1652.19
  5912.7 1660.54  5922.7 1661.42  6013.2 1662.33  6073.5 1660.96  6109.4 1661.81
#Mann= 11 ,-1 , 0
  3184.8    .035       0  3631.2     .07       0  3725.2    .035       0
    3977     .07       0  4167.6    .035       0  4983.1     .07       0
  4992.2    .035       0  5096.6    .035       0  5196.7     .07       0
  5482.8    .035       0    5746     .07       0
Bank Sta=4983.1,4992.2
XS Rating Curve= 0 ,0
Exp/Cntr=0.3,0.1

Type RM Length L Ch R = 1 ,16169   ,632,632,632
BEGIN DESCRIPTION:
Mapping XS 2ae136ef
END DESCRIPTION:
XS GIS Cut Line= 3
      1573273.67      6883264.02      1574836.14      6883125.14
      1575890.43      6882856.14
#Sta/Elev= 30
  3411.9 1660.58  3989.3 1654.63  4284.3 1649.99  4417.2 1646.36  4487.5 1643.21
  4626.1 1642.22  4678.2 1641.15  4738.4 1642.36  4992.9 1640.65  5015.1 1640.07
  5015.6 1639.57  5026.2 1640.07  5029.4 1640.42  5247.7 1640.63  5340.6 1642.47
  5381.9 1641.63  5518.1 1642.88  5650.2 1642.19  5793.8 1646.34    5799 1645.55
  5834.7 1646.36  5839.9 1645.31  5880.7  1647.1  5897.9 1648.89  5916.4 1654.32
  5921.6 1654.03  5928.8 1657.39  5974.5 1658.37  5988.4 1658.51  6068.6 1659.21
#Mann= 9 ,-1 , 0
  3411.9    .035       0  4284.3     .07       0  4626.1    .035       0
  4992.9     .07       0  5015.1     .07       0  5026.2     .07       0
  5029.4    .035       0  5974.5     .07       0  5988.4    .035       0
Bank Sta=5015.1,5026.2
XS Rating Curve= 0 ,0
Exp/Cntr=0.3,0.1

Type RM Length L Ch R = 1 ,15537   ,956,956,956
BEGIN DESCRIPTION:
Mapping XS 598ae9b6
END DESCRIPTION:
XS GIS Cut Line= 4
      1573354.39      6883845.33      1574656.46      6883663.04
      1575088.75      6883517.21      1575821.58      6882971.48
#Sta/Elev= 30
  3687.2 1659.44  3779.9 1657.29  3917.7 1652.64  4208.4 1653.64  4475.1 1651.73
  4519.6 1651.21  4641.8 1649.81  4753.2 1647.24  4818.7  1645.4  4843.3 1643.93
  4916.7 1641.29  5015.8 1637.14  5016.3 1636.64  5027.2 1637.14  5035.4  1638.1
  5104.7 1638.52  5483.3 1641.52  5698.1 1640.45  5783.6 1641.81  5804.5 1640.79
  6140.2 1644.93  6148.6 1648.01  6154.8 1652.38  6163.2 1656.62  6169.4 1658.72
  6176.7 1659.28  6269.5  1658.1  6298.8 1659.19  6357.2 1658.88  6371.9 1658.66
#Mann= 10 ,-1 , 0
  3687.2    .035       0  4475.1     .07       0  4519.6    .035       0
  4753.2     .07       0  4843.3    .035       0  4916.7     .07       0
  5015.8     .07       0  5027.2     .07       0  5104.7    .035       0
  6357.2    .063       0
Bank Sta=5015.8,5027.2
XS Rating Curve= 0 ,0
Exp/Cntr=0.3,0.1

Type RM Length L Ch R = 1 ,14581   ,900,900,900
BEGIN DESCRIPTION:
Mapping XS a622d2ce
END DESCRIPTION:
XS GIS Cut Line= 4
      1573547.07        6884637.      1574812.71      6884402.63
      1575198.12      6884178.67      1575807.49      6883038.06
#Sta/Elev= 30
  3720.3 1657.46  3884.8  1655.3  4070.4  1651.8  4318.2 1651.32  4450.3 1649.36
  4465.5 1648.83    4582 1645.89  4651.3 1643.16  4775.9 1636.74  4847.1 1635.36
  4899.3 1637.57  4958.9  1635.8  4973.4  1633.1  4973.9  1632.6  4985.1  1633.1
  5056.4 1636.97  5230.6 1638.65  5262.1 1637.17  5363.9 1637.29  5524.3 1640.08
  5873.5 1640.55  5886.1 1639.54    6056 1642.45  6447.2 1645.12  6576.3 1645.88
  6587.7 1653.14  6598.3 1657.18  6607.7 1658.06  6691.8 1660.23  6746.4 1659.27
#Mann= 10 ,-1 , 0
  3720.3     .07       0  3884.8    .035       0  4450.3     .07       0
  4465.5    .035       0    4582     .07       0  4651.3    .035       0
  4973.4    .035       0  4985.1    .035       0  6447.2    .063       0
  6607.7    .035       0
Bank Sta=4973.4,4985.1
XS Rating Curve= 0 ,0
Exp/Cntr=0.3,0.1

Type RM Length L Ch R = 1 ,13681   ,266,266,266
BEGIN DESCRIPTION:
MULBERRY CREEK TRIBUTARY 4 10.0
END DESCRIPTION:
XS GIS Cut Line= 4
      1573390.85      6884850.55        1574555.        6885138.
       1575307.5      6884376.58      1575580.01      6883912.98
#Sta/Elev= 30
  3806.6  1657.7  4449.5 1647.42  4748.2  1645.8  4768.8 1644.06  4799.7 1636.45
  4830.6 1633.39  4840.9 1629.67  4865.9 1629.53  4866.4 1629.03  4877.7 1629.53
  4910.8 1629.61  4995.4 1629.71  5012.8 1630.24    5034 1633.67  5126.5 1634.57
  5147.1 1635.65  5168.4 1633.59  5189.5 1634.47    5232 1632.34  5288.5 1635.34
  5345.1    1633  5387.5 1636.05  5437.1 1636.81  5649.2 1637.62  5734.1 1635.76
  5858.9    1637  6046.5 1638.41  6094.6 1638.83  6242.3    1639    6614 1641.41
#Mann= 10 ,-1 , 0
  3806.6    .035       0  4748.2     .07       0  4865.9    .033       0
  4877.7     .07       0  4910.8    .033       0  5126.5    .035       0
  5858.9     .07       0  6046.5    .035       0  6094.6     .07       0
  6242.3    .035       0
Bank Sta=4865.9,4877.7
XS Rating Curve= 0 ,0
Exp/Cntr=0.3,0.1
