--- WEAVER SPRINGS CREEK TRIB 1.prj (project) ---

Proj Title=WEAVER SPRINGS CREEK TRIB 1 Base Level Engineering
Current Plan=p01
Default Exp/Contr=0.3,0.1
English Units
Geom File=g01
Flow File=f01
Plan File=p01
Y Axis Title=Elevation
X Axis Title(PF)=Main Channel Distance
X Axis Title(XS)=Station
BEGIN DESCRIPTION:
WEAVER SPRINGS CREEK TRIB 1
END DESCRIPTION:
DSS Export Rating Curves= 0
DSS Export Rating Curve Sorted= 0
DSS Export Volume Flow Curves= 0
DXF OffsetX= 0
DXF OffsetY= 0
DXF ScaleX= 1
DXF ScaleY= 10

--- WEAVER SPRINGS CREEK TRIB 1.p01 (plan) ---

Plan Title=Multiple Run
Short Identifier=Multiple
Geom File=g01
Flow File=f01
Subcritical Flow
K Sum by GR= 0
Std Step Tol= 0.01
Critical Tol= 0.01
Num of Std Step Trials= 20
Max Error Tol= 0.3
Flow Tol Ratio= 0.001
Split Flow NTrial= 30
Split Flow Tol= 0.02
Split Flow Ratio= 0.02
Log Output Level= 0
Friction Slope Method= 1
Unsteady Friction Slope Method= 2
Unsteady Bridges Friction Slope Method= 1
Parabolic Critical Depth
Global Vel Dist=  1 , 1 , 1
Global Log Level= 0
CheckData=True
Encroach Param= -1, 0, 0, 0
BEGIN DESCRIPTION:
Multiple Run
END DESCRIPTION:

--- WEAVER SPRINGS CREEK TRIB 1.f01 (steady flow) ---

Flow Title=Multiple
Program Version=4.10
Number of Profiles= 7
Profile Names=10-year,25-year,50-year,1pct_min,100-year,1pct_plu,500-year
River Rch & RM=WEAVER SPRINGS C,Reach-1         ,29073
     523     770     986     628    1254    2502    2051
River Rch & RM=WEAVER SPRINGS C,Reach-1         ,24296
     647     961    1239     794    1584    3160    2619
River Rch & RM=WEAVER SPRINGS C,Reach-1         ,18985
    1096    1671    2191    1425    2843    5673    4852
River Rch & RM=WEAVER SPRINGS C,Reach-1         ,16845
    1299    1994    2627    1716    3424    6831    5892
River Rch & RM=WEAVER SPRINGS C,Reach-1         ,15211
    1323    2029    2670    1742    3475    6934    5965
River Rch & RM=WEAVER SPRINGS C,Reach-1         ,10805
    1424    2188    2882    1882    3755    7491    6455
River Rch & RM=WEAVER SPRINGS C,Reach-1         ,8032
    1455    2230    2935    1913    3817    7616    6542
River Rch & RM=WEAVER SPRINGS C,Reach-1         ,1775
    1534    2356    3104    2026    4042    8065    6944
Boundary for River Rch & Prof#=WEAVER SPRINGS C,Reach-1         , 1
Up Type= 0
Dn Type= 3
Dn Slope=0.00796
Boundary for River Rch & Prof#=WEAVER SPRINGS C,Reach-1         , 2
Up Type= 0
Dn Type= 3
Dn Slope=0.00796
Boundary for River Rch & Prof#=WEAVER SPRINGS C,Reach-1         , 3
Up Type= 0
Dn Type= 3
Dn Slope=0.00796
Boundary for River Rch & Prof#=WEAVER SPRINGS C,Reach-1         , 4
Up Type= 0
Dn Type= 3
Dn Slope=0.00796
Boundary for River Rch & Prof#=WEAVER SPRINGS C,Reach-1         , 5
Up Type= 0
Dn Type= 3
Dn Slope=0.00796
Boundary for River Rch & Prof#=WEAVER SPRINGS C,Reach-1         , 6
Up Type= 0
Dn Type= 3
Dn Slope=0.00796
Boundary for River Rch & Prof#=WEAVER SPRINGS C,Reach-1         , 7
Up Type= 0
Dn Type= 3
Dn Slope=0.00796
DSS Import GetInterval= 0
DSS Import GetPeak= 0
DSS Import FillOption= 0

--- WEAVER SPRINGS CREEK TRIB 1.g01 (geometry) ---

Geom Title=Existing Conditions
Program Version=4.10

River Reach=WEAVER SPRINGS C,Reach-1
Reach XY= 30
        1441955.        6833188.      1442715.48      6832588.93
      1444285.01      6832988.06      1444903.54      6832884.46
      1445534.97      6832387.55      1445775.05      6832638.21
      1446353.38      6832441.12      1446965.27      6832887.03
       1447893.3      6832788.99      1448752.32      6833482.58
      1449484.97      6833587.94      1450956.58      6832441.67
      1451399.07      6832585.77      1452204.96      6832145.52
      1453057.45      6832282.54      1453251.96      6831739.42
      1452606.74      6830994.16      1452806.64      6830641.09
      1453089.04      6830787.11      1453838.95      6830455.05
      1453655.81      6829899.94      1454038.24      6829404.43
      1454724.88      6828937.93      1456399.07      6829235.76
      1456949.18      6828740.28      1456951.84      6828096.34
      1456307.14      6827243.97      1457502.77       6825582.1
      1457010.54      6824635.63        1458205.        6823738.

Type RM Length L Ch R = 1 ,29073   ,394,394,394
BEGIN DESCRIPTION:
WEAVER SPRINGS CREEK TRIB 1 50.0
END DESCRIPTION:
XS GIS Cut Line= 3
      1442152.44      6833431.03      1442141.94      6833138.32
        1441805.      6832842.45
#Sta/Elev= 30
  4707.1 2430.76  4711.1 2430.76  4770.2 2411.91  4775.2  2413.8  4780.2 2411.12
  4800.2 2405.85  4840.2 2401.12  4880.2 2394.56  4900.3 2388.98  4940.3 2383.53
  4950.3 2381.37  4960.3  2377.9  4980.3 2359.57  4990.3 2351.75  5003.3 2348.16
  5003.6 2347.66  5007.3 2348.16    5012 2349.66  5033.8 2353.19  5040.4 2355.34
  5111.6 2358.02  5132.5 2357.95  5260.6 2367.16  5324.1 2373.97  5338.4 2376.18
  5381.1 2385.29  5416.2 2394.64  5422.8 2397.44  5444.7 2402.34  5448.4 2405.05
#Mann= 3 ,-1 , 0
  4707.1     .07       0  5003.3     .07       0  5007.3     .16       0
Bank Sta=5003.3,5007.3
XS Rating Curve= 0 ,0
Exp/Cntr=0.3,0.1

Type RM Length L Ch R = 1 ,28679   ,410,410,410
BEGIN DESCRIPTION:
Mapping XS 37b88874
END DESCRIPTION:
XS GIS Cut Line= 3
      1442584.17      6833341.95       1442403.6      6832904.41
      1441941.83      6832626.66
#Sta/Elev= 30
    4411 2443.34  4450.6 2441.25  4469.2 2434.78  4474.6 2435.15  4480.2 2430.64
  4498.5 2421.94  4503.9 2421.75  4551.7  2404.9  4704.5 2377.97  4711.5 2378.12
  4735.4 2371.68  4740.9 2372.05  4788.7 2357.32  4804.7 2355.31  4865.9    2352
  4988.8 2351.03  5019.9 2342.89  5032.4 2342.26  5032.7 2341.76  5036.4 2342.26
  5047.1  2342.6  5056.8 2345.93  5078.2 2357.27  5092.8 2361.72  5179.2 2371.26
  5258.8 2387.57  5326.1 2406.32    5354  2416.4  5390.9 2433.13  5423.2 2441.56
#Mann= 4 ,-1 , 0
    4411     .07       0  4704.5     .16       0  5032.4     .07       0
  5036.4     .16       0
Bank Sta=5032.4,5036.4
XS Rating Curve= 0 ,0
Exp/Cntr=0.3,0.1

Type RM Length L Ch R = 1 ,28269   ,584,584,584
BEGIN DESCRIPTION:
Mapping XS b6f909a2
END DESCRIPTION:
XS GIS Cut Line= 3
      1443018.16      6833272.44      1442625.82      6832675.25
      1442266.44       6832492.1
#Sta/Elev= 30
  4279.4 2447.01  4343.7 2445.86  4379.9 2442.26  4406.9 2425.29  4455.6 2406.61
    4482 2397.36  4515.4 2385.29  4575.1 2371.47  4608.8 2364.47  4675.1 2356.64
  4783.6 2350.83  4978.7 2345.79  4996.4 2342.94  5004.1 2338.14  5004.3 2337.64
  5008.1 2338.14  5060.8 2341.46    5083 2348.46  5088.6 2353.87  5105.2 2359.25
  5110.9 2366.26  5127.5 2371.18  5133.1  2376.9  5139.7 2379.03  5155.3 2384.39
  5297.9 2406.02  5355.5 2423.95  5377.7 2428.89  5394.3 2427.72  5397.3 2429.76
#Mann= 7 ,-1 , 0
  4279.4     .07       0  4455.6     .16       0    4482     .07       0
  4575.1     .16       0  5004.1     .07       0  5008.1     .16       0
  5139.7     .07       0
Bank Sta=5004.1,5008.1
XS Rating Curve= 0 ,0
Exp/Cntr=0.3,0.1

Type RM Length L Ch R = 1 ,27685   ,321,321,321
BEGIN DESCRIPTION:
Mapping XS 967a19d7
END DESCRIPTION:
XS GIS Cut Line= 3
      1443066.79      6833272.44      1443118.88      6832741.22
      1443000.84      6831942.76
#Sta/Elev= 30
  4463.3 2446.68  4568.2 2443.92  4618.5 2436.67  4648.6  2425.4  4668.7 2414.09
  4697.5 2404.05    4799  2384.7  4829.5 2381.19  4849.6 2376.34  4864.8  2369.3
  4905.5 2348.63  4910.5 2350.03    4930 2341.35  4960.1 2340.12    4978 2330.67
  4978.3 2330.17  4982.5 2330.67  4996.2 2333.69  5030.6 2334.71  5050.9 2339.67
    5196 2341.52  5364.2 2348.89  5414.8 2354.62  5469.2 2365.01  5505.8 2378.49
  5637.2 2404.69  5667.5 2413.52    5718 2434.61  5748.4 2441.58  5804.2 2445.88
#Mann= 4 ,-1 , 0
  4463.3     .07       0  4864.8     .16       0    4978     .07       0
  4982.5     .16       0
Bank Sta=4978,4982.5
XS Rating Curve= 0 ,0
Exp/Cntr=0.3,0.1

Type RM Length L Ch R = 1 ,27364   ,404,404,404
BEGIN DESCRIPTION:
Mapping XS 11519a1f
END DESCRIPTION:
XS GIS Cut Line= 3
      1443108.45       6833321.1      1443414.01      6832737.75
      1443587.62      6831973.86
#Sta/Elev= 30
  4350.7 2446.15  4409.5    2445  4455.8 2441.16  4489.7 2428.24  4566.3    2408
  4670.3 2392.17  4720.7 2381.32  4737.2  2381.9  4742.8 2380.03  4759.2 2382.08
  4764.9 2380.18  4869.6 2376.42  4891.6  2368.2  4932.2 2345.08  4952.2 2335.09
  4986.4 2330.02  4999.6 2324.76    5000 2324.26  5004.2 2324.76  5006.3 2328.02
  5011.7 2328.02  5035.4 2336.49  5162.8 2334.78    5218 2336.27  5443.6 2349.79
  5480.7 2357.31  5577.9 2385.92  5712.3  2436.2  5737.1 2443.26  5792.6 2450.23
#Mann= 5 ,-1 , 0
  4350.7     .16       0  4409.5     .07       0  4932.2     .16       0
  4999.6     .07       0  5004.2     .16       0
Bank Sta=4999.6,5004.2
XS Rating Curve= 0 ,0
Exp/Cntr=0.3,0.1

Type RM Length L Ch R = 1 ,26960   ,296,296,296
BEGIN DESCRIPTION:
Mapping XS 1bc3d40a
END DESCRIPTION:
XS GIS Cut Line= 3
      1443149.24      6833377.52      1443709.15      6832887.92
      1443911.71      6832241.29
#Sta/Elev= 30
  4046.2 2442.79  4106.6 2434.93  4148.9 2426.61    4220  2405.2  4297.9 2389.63
  4340.6 2375.52  4361.5 2377.19  4369.1 2372.92  4375.7 2375.26  4383.3  2372.3
  4418.4    2376  4432.7 2370.16  4439.3 2372.63  4446.9 2368.97  4453.5  2370.9
  4496.2 2363.91    4539 2349.36  4679.8    2340  4864.1 2328.39  4905.2 2329.76
    4968 2324.98  4986.3 2320.46  4986.6 2319.96    4991 2320.46    5010 2329.03
  5091.2 2330.63  5291.1 2400.33  5334.8  2419.3  5431.4 2444.46  5467.6 2447.64
#Mann= 5 ,-1 , 0
  4046.2     .16       0  4106.6     .07       0  4679.8     .16       0
  4986.3     .07       0    4991     .16       0
Bank Sta=4986.3,4991
XS Rating Curve= 0 ,0
Exp/Cntr=0.3,0.1

Type RM Length L Ch R = 1 ,26664   ,306,306,306
BEGIN DESCRIPTION:
Mapping XS e53a533c
END DESCRIPTION:
XS GIS Cut Line= 3
      1443901.86      6833710.84      1443977.38      6832973.86
      1444115.21      6832412.16
#Sta/Elev= 30
  4126.2 2443.61  4169.3 2431.78  4205.2 2415.16  4229.6 2408.02  4340.2 2395.57
  4440.7 2378.42  4480.9 2362.66  4498.1 2352.16  4521.1 2346.04  4552.3 2343.54
  4641.7 2337.67  4878.1 2331.54  4966.4 2321.14  4973.5 2317.83  4973.9 2317.33
  4978.5 2317.83    5008 2325.31  5132.7 2325.62  5151.1 2329.72  5169.1 2337.24
  5174.3  2336.7  5210.7 2357.01  5252.3 2375.03  5257.4  2375.1  5293.9 2391.78
  5340.6 2407.82    5377 2426.44  5382.2 2425.79  5408.5 2443.67  5445.4 2447.12
#Mann= 4 ,-1 , 0
  4126.2     .07       0  4552.3     .16       0  4973.5     .07       0
  4978.5     .16       0
Bank Sta=4973.5,4978.5
XS Rating Curve= 0 ,0
Exp/Cntr=0.3,0.1

Type RM Length L Ch R = 1 ,26358   ,516,516,516
BEGIN DESCRIPTION:
Mapping XS ba920654
END DESCRIPTION:
XS GIS Cut Line= 3
      1444091.96      6833848.87      1444245.61      6833005.11
       1444175.3      6832424.39
#Sta/Elev= 30
  4125.6 2449.96    4144 2449.11  4171.3 2444.82  4224.7 2420.48  4229.7 2420.41
    4278 2402.95  4283.1 2404.27  4289.1 2399.53  4336.4 2384.26  4448.1 2365.63
  4642.2 2345.97  4797.3 2333.86    4960 2324.77    5008 2315.09  5008.4 2314.59
    5013 2315.09  5020.6 2317.98  5042.1  2318.5  5093.7 2321.65  5161.6 2317.63
  5181.8 2321.76  5232.1 2323.52  5302.7 2334.34  5332.9 2346.04  5360.4 2367.03
  5365.4 2367.43  5373.2 2372.43    5494 2412.21  5544.4 2433.11  5568.2 2437.64
#Mann= 7 ,-1 , 0
  4125.6     .16       0    4144     .07       0  4642.2     .16       0
    5008     .07       0    5013     .16       0  5042.1     .07       0
  5093.7     .16       0
Bank Sta=5008,5013
XS Rating Curve= 0 ,0
Exp/Cntr=0.3,0.1

Type RM Length L Ch R = 1 ,25842   ,350,350,350
BEGIN DESCRIPTION:
Mapping XS 28e9befa
END DESCRIPTION:
XS GIS Cut Line= 4
      1444323.74      6833799.38      1444690.92        6832940.
      1444680.51      6832851.46      1444295.54      6832162.16
#Sta/Elev= 30
  4013.3 2447.12  4077.4 2445.01  4106.4 2437.89  4188.8 2407.45  4243.2 2400.93
  4297.5 2388.41  4411.4 2376.92  4440.4 2366.84  4493.3 2341.84  4657.9 2328.37
  4792.6 2317.67  4816.2 2317.86  4821.6 2321.11  4866.7 2319.12  5017.7 2308.82
  5018.1 2308.32  5022.9 2308.82  5052.4 2314.83  5185.7 2319.67  5337.6 2332.75
  5430.8 2342.98  5507.3 2353.15  5534.7 2359.79  5550.7 2359.82  5594.1 2370.71
  5625.1 2373.99  5712.9 2400.98  5788.1 2433.19  5808.4 2442.78  5826.5 2446.06
#Mann= 9 ,-1 , 0
  4013.3     .07       0  4657.9     .16       0  4866.7     .07       0
  5017.7     .07       0  5022.9     .07       0  5185.7     .16       0
  5337.6     .07       0  5430.8     .16       0  5788.1     .07       0
Bank Sta=5017.7,5022.9
XS Rating Curve= 0 ,0
Exp/Cntr=0.3,0.1

Type RM Length L Ch R = 1 ,25492   ,635,635,635
BEGIN DESCRIPTION:
WEAVER SPRINGS CREEK TRIB 1 42.0
END DESCRIPTION:
XS GIS Cut Line= 3
      1445263.08      6833560.65      1444998.51      6832794.76
      1444482.93      6832181.76
#Sta/Elev= 30
  4189.7 2445.42  4199.8 2445.08  4224.2 2442.63  4260.8 2428.84  4277.1  2418.9
  4298.3 2410.19  4416.7 2377.92  4442.6 2365.13    4505 2350.44  4749.2  2321.1
    4859 2313.85  4978.7 2310.44  4993.4 2308.68  4997.7 2306.09  5014.9 2305.15
  5025.9 2304.67  5026.3 2304.17  5031.2 2304.67  5113.4 2307.77  5163.1 2312.62
  5202.6 2314.07  5361.4 2323.99  5386.1 2325.43  5517.1 2336.99  5546.3 2341.44
  5560.6 2346.23  5617.8 2373.82  5681.5 2384.61  5759.6 2401.27    5801 2416.59
#Mann= 11 ,-1 , 0
  4189.7     .16       0  4199.8     .07       0  4978.7     .16       0
  5014.9     .07       0  5025.9     .07       0  5031.2     .07       0
  5163.1     .16       0  5202.6     .07       0  5361.4     .16       0
  5386.1     .07       0  5517.1     .16       0
Bank Sta=5025.9,5031.2
XS Rating Curve= 0 ,0
Exp/Cntr=0.3,0.1

Type RM Length L Ch R = 1 ,24857   ,561,561,561
BEGIN DESCRIPTION:
WEAVER SPRINGS CREEK TRIB 1 41.0
END DESCRIPTION:
XS GIS Cut Line= 3
        1445405.      6833238.03        1445405.        6832438.
      1445005.01      6832038.01
#Sta/Elev= 30
  4204.7 2381.82  4224.7 2375.97  4274.7 2348.09  4284.7 2343.42  4304.7 2336.99
  4344.7 2332.06  4384.7 2324.23  4449.3 2318.69  4604.8 2307.31  4684.7 2302.58
  4729.6 2303.31  4784.7    2304  4934.7 2299.63  4982.1 2295.49  4982.5 2294.99
  4987.4 2295.49  5008.3 2297.08  5018.9 2301.12    5033 2301.85  5075.4 2307.68
  5216.9 2312.99  5370.5 2323.71  5422.2 2331.27  5443.1 2334.05  5471.4 2341.55
  5499.7 2355.88  5513.8  2365.5    5528 2371.58  5556.3 2378.78  5570.4 2380.67
#Mann= 8 ,-1 , 0
  4204.7     .07       0  4449.3     .16       0  4604.8     .07       0
  4729.6     .16       0  4982.1     .07       0  4987.4     .16       0
  5370.5     .07       0  5422.2     .16       0
Bank Sta=4982.1,4987.4
XS Rating Curve= 0 ,0
Exp/Cntr=0.3,0.1

Type RM Length L Ch R = 1 ,24296   ,146,146,146
BEGIN DESCRIPTION:
WEAVER SPRINGS CREEK TRIB 1 40.0
END DESCRIPTION:
XS GIS Cut Line= 3
      1445858.78      6833457.81      1445825.04      6832638.61
      1445821.15      6831693.22
#Sta/Elev= 30
  4180.1 2420.19    4270  2398.3    4340 2379.56  4350.1 2375.92  4370.1 2364.46
  4394.3 2353.27  4400.1 2348.45  4420.1 2340.11  4430.1 2337.75  4580.3 2320.36
  4660.3 2313.14  4900.5 2298.79  4910.5 2297.56  4940.6 2288.75  4960.5 2286.27
  4961.4 2286.23  4994.9 2285.05  4995.4 2284.55  5000.7 2285.05  5150.6  2291.3
  5190.6 2297.61  5305.6 2308.11  5510.6 2323.95  5680.6 2334.37  5740.4 2344.23
  5780.6 2352.57  5840.6 2372.06  5860.6 2376.75  5890.6 2382.08  5945.4 2388.58
#Mann= 7 ,-1 , 0
  4180.1     .07       0  4960.5     .16       0  4961.4     .07       0
  4994.9     .07       0  5000.7     .07       0  5305.6     .16       0
  5740.4     .07       0
Bank Sta=4994.9,5000.7
XS Rating Curve= 0 ,0
Exp/Cntr=0.3,0.1

Type RM Length L Ch R = 1 ,24150   ,713,713,713
BEGIN DESCRIPTION:
WEAVER SPRINGS CREEK TRIB 1 39.0
END DESCRIPTION:
XS GIS Cut Line= 4
      1445967.44      6833444.51      1445954.83       6832587.6
      1445954.56      6832341.89      1446224.25      6831918.02
#Sta/Elev= 30
    4143 2435.49  4319.5 2381.16  4379.5 2342.99  4399.5 2334.57  4419.5 2329.51
  4599.6 2312.53  4799.6 2300.44  4929.6  2296.9  4986.7 2289.57  4987.2 2289.07
  4992.5 2289.57  5109.6 2294.64  5313.6 2310.97  5386.4 2323.85  5429.1 2336.93
  5474.5 2357.67  5501.6 2374.02  5548.1 2391.32  5574.4 2401.43  5589.6 2404.45
  5595.6 2408.33  5604.9 2409.65  5610.8 2413.95    5626 2416.42    5632 2421.56
  5662.5 2427.68  5668.4 2432.04  5683.6  2432.3  5704.8 2439.51  5748.1 2442.89
#Mann= 5 ,-1 , 0
    4143     .07       0  4986.7     .07       0  4992.5     .07       0
  5429.1     .16       0  5548.1     .07       0
Bank Sta=4986.7,4992.5
XS Rating Curve= 0 ,0
Exp/Cntr=0.3,0.1

Type RM Length L Ch R = 1 ,23437   ,329,329,329
BEGIN DESCRIPTION:
WEAVER SPRINGS CREEK TRIB 1 38.0
END DESCRIPTION:
XS GIS Cut Line= 3
      1446122.16      6833439.32      1446510.85      6832636.46
      1446655.01      6832137.98
#Sta/Elev= 30
    4108 2386.53  4142.8 2377.97  4148.6 2373.44  4187.2 2358.25  4231.7 2350.96
  4306.7 2335.42    4365 2325.33  4431.7 2316.78  4553.9 2305.03  4763.8 2293.25
  4813.8  2292.2  4950.2 2288.65  4975.5 2275.99  4975.9 2275.49  4981.3 2275.99
  4987.2 2280.01    5040 2280.06  5060.9 2282.59  5112.9 2284.22  5139.9 2290.49
  5178.7 2295.72  5212.4 2303.92  5251.2 2308.86  5357.2 2339.15  5362.7 2342.95
    5396 2355.33  5435.6 2376.26  5502.1 2403.31  5516.3 2412.15  5518.9 2412.15
#Mann= 6 ,-1 , 0
    4108     .07       0  4553.9     .16       0  4763.8     .07       0
  4813.8     .16       0  4975.5     .07       0  4981.3     .16       0
Bank Sta=4975.5,4981.3
XS Rating Curve= 0 ,0
Exp/Cntr=0.3,0.1

Type RM Length L Ch R = 1 ,23108   ,307,307,307
BEGIN DESCRIPTION:
WEAVER SPRINGS CREEK TRIB 1 37.0
END DESCRIPTION:
XS GIS Cut Line= 3
      1446266.82      6833486.07        1446805.        6832638.
      1446820.65      6832132.66
#Sta/Elev= 30
  3995.2 2355.61  4115.2    2332    4188 2322.59  4217.9 2321.08  4305.7 2311.56
  4397.3 2304.92  4488.6 2300.93    4514 2299.41    4637    2300  4673.5  2297.1
  4709.9 2289.93  4753.3 2286.62  4803.9 2283.47  4840.4 2285.41    4892 2280.01
  4955.6 2278.94  4986.1 2276.56  4996.7 2272.81  5006.7 2271.76  5007.2 2271.26
  5012.6 2271.76  5059.6 2283.66  5162.9 2291.06  5259.7  2315.2  5319.8 2336.62
  5439.8 2394.72  5479.5 2411.17  5482.5 2410.09  5484.5 2409.37  5505.2 2420.06
#Mann= 7 ,-1 , 0
  3995.2     .07       0  4305.7     .16       0  4488.6     .07       0
  4753.3     .16       0  5006.7     .07       0  5012.6     .16       0
  5482.5     .07       0
Bank Sta=5006.7,5012.6
XS Rating Curve= 0 ,0
Exp/Cntr=0.3,0.1

Type RM Length L Ch R = 1 ,22801   ,488,488,488
BEGIN DESCRIPTION:
WEAVER SPRINGS CREEK TRIB 1 36.0
END DESCRIPTION:
XS GIS Cut Line= 3
      1446403.99      6833580.23      1446956.23      6832884.57
       1447500.2      6831916.43
#Sta/Elev= 30
  4111.8 2333.87  4151.7 2330.86  4313.5 2316.93  4565.9 2302.16  4620.2 2299.67
    4791 2291.16  4890.3 2290.03  4960.8  2285.3  4975.2 2283.52    4992 2267.83
  4992.5 2267.33  4997.9 2267.83    5042 2275.08  5156.7 2276.62  5296.8 2283.97
    5453 2294.49    5599 2301.09  5604.7 2300.08  5723.3 2304.56  5798.6  2311.3
  5847.7 2318.87  5922.9 2339.45  5928.6 2339.46  5944.6 2345.23  5950.3 2345.66
    5994 2369.98  6016.9  2378.9  6062.8 2393.44  6068.9 2396.79  6110.5  2407.4
#Mann= 6 ,-1 , 0
  4111.8     .07       0  4151.7     .16       0  4565.9     .07       0
  4620.2     .16       0    4992     .07       0  4997.9     .16       0
Bank Sta=4992,4997.9
XS Rating Curve= 0 ,0
Exp/Cntr=0.3,0.1

Type RM Length L Ch R = 1 ,22313   ,560,560,560
BEGIN DESCRIPTION:
WEAVER SPRINGS CREEK TRIB 1 35.0
END DESCRIPTION:
XS GIS Cut Line= 3
      1446779.85      6833848.47      1447394.45      6832945.68
      1447592.35      6831935.31
#Sta/Elev= 30
  3900.5 2339.18  3933.8  2329.6  3990.7 2325.91  4111.2 2314.37  4389.7 2297.92
  4436.6 2294.67  4574.2 2291.03  4622.3 2287.83    4760 2276.31  4954.4 2274.11
  4969.3 2273.01  4984.3 2266.32  4997.5 2262.82    4998 2262.32  5003.4 2262.82
  5051.4 2270.98  5229.7 2275.52  5440.7 2292.04  5479.4 2293.63  5698.1 2316.56
  5764.7 2326.42  5846.2 2342.79  5866.6 2349.95  5904.1 2367.33  5909.2 2367.15
  5937.9 2378.48  5955.6 2383.93  5960.7 2383.31  6007.1  2399.1  6022.2 2401.55
#Mann= 6 ,-1 , 0
  3900.5     .07       0  4111.2     .16       0  4389.7     .07       0
  4622.3     .16       0  4997.5     .07       0  5003.4     .16       0
Bank Sta=4997.5,5003.4
XS Rating Curve= 0 ,0
Exp/Cntr=0.3,0.1

Type RM Length L Ch R = 1 ,21753   ,363,363,363
BEGIN DESCRIPTION:
WEAVER SPRINGS CREEK TRIB 1 34.0
END DESCRIPTION:
XS GIS Cut Line= 3
      1446915.28      6833997.76        1447905.        6832788.
      1447818.23      6832241.88
#Sta/Elev= 30
  3444.1 2348.63  3450.9 2348.21  3457.4 2341.82  3465.3 2341.32  3471.7 2337.28
  3500.4 2330.76    3599 2318.15  3714.3 2309.15  4041.6  2291.6  4382.8 2274.41
  4599.6  2268.6  4730.1 2269.45  4851.8 2266.49  4976.1 2257.04  4976.6 2256.54
  4982.2 2257.04  4993.5 2260.04  5003.9 2268.07  5017.3 2271.42  5244.4  2289.5
  5289.7 2295.53  5351.4 2313.86  5381.8 2315.58  5412.2 2324.39  5445.6 2342.84
  5479.7 2364.02  5493.2 2374.87  5503.3 2377.85  5533.7 2383.31  5560.1 2383.97
#Mann= 11 ,-1 , 0
  3444.1     .07       0    3599     .16       0  4041.6     .07       0
  4382.8     .16       0  4599.6     .07       0  4851.8     .16       0
  4976.1     .07       0  4982.2     .16       0  5244.4     .07       0
  5445.6     .16       0  5479.7     .07       0
Bank Sta=4976.1,4982.2
XS Rating Curve= 0 ,0
Exp/Cntr=0.3,0.1

Type RM Length L Ch R = 1 ,21390   ,522,522,522
BEGIN DESCRIPTION:
WEAVER SPRINGS CREEK TRIB 1 33.0
END DESCRIPTION:
XS GIS Cut Line= 3
      1447547.12      6834393.63      1448115.19      6832987.55
      1448625.25      6832284.23
#Sta/Elev= 30
  3483.5 2412.67  3565.1 2383.16  3570.9 2377.55  3576.3 2378.89    3595 2368.58
  3600.4 2371.09  3624.5 2356.54  3702.3 2335.86  3839.2 2307.98  3970.2 2295.61
  4048.6 2289.58  4528.5 2270.72  4586.4 2268.71  4690.8 2265.75  4805.4 2258.61
  4823.8 2262.39  4955.2 2262.06    4987 2254.49  4987.5 2253.99  4993.2 2254.49
  5042.5  2256.5  5092.7 2267.63  5335.5 2280.56  5493.6 2297.36    5580 2321.04
    5637 2331.85  5708.1 2375.56  5787.8 2404.26  5851.8 2434.65  5868.8 2437.12
#Mann= 8 ,-1 , 0
  3483.5     .07       0  3970.2     .16       0  4048.6     .07       0
  4528.5     .16       0  4586.4     .07       0  4690.8     .16       0
    4987     .07       0  4993.2     .16       0
Bank Sta=4987,4993.2
XS Rating Curve= 0 ,0
Exp/Cntr=0.3,0.1

Type RM Length L Ch R = 1 ,20868   ,440,440,440
BEGIN DESCRIPTION:
WEAVER SPRINGS CREEK TRIB 1 32.0
END DESCRIPTION:
XS GIS Cut Line= 3
      1447844.03       6834419.6        1448505.        6833188.
      1448922.14      6832325.87
#Sta/Elev= 30
  3602.2 2363.94  3661.8  2344.1  3728.9 2326.26  3847.7 2305.68  3957.3 2292.29
  4077.5 2285.49    4092    2282  4143.3 2282.69  4252.9  2276.8    4633 2267.93
  4691.1 2263.51  4799.8 2257.89  4904.1 2256.85  4926.1 2255.02  4942.3 2250.39
  4982.9 2248.76  4983.4 2248.26  4989.5 2248.76  5255.5 2267.26  5358.4 2278.03
  5584.3 2310.17  5629.5 2320.97  5680.2 2340.23  5697.2 2343.98  5777.6 2378.23
  5810.2 2389.04  5838.3 2403.51  5915.1 2434.88  5928.7 2440.58  5957.7 2442.31
#Mann= 7 ,-1 , 0
  3602.2     .07       0    4633     .16       0  4691.1     .07       0
  4799.8     .16       0  4982.9     .07       0  4989.5     .16       0
  5915.1     .07       0
Bank Sta=4982.9,4989.5
XS Rating Curve= 0 ,0
Exp/Cntr=0.3,0.1

Type RM Length L Ch R = 1 ,20428   ,481,481,481
BEGIN DESCRIPTION:
WEAVER SPRINGS CREEK TRIB 1 31.0
END DESCRIPTION:
XS GIS Cut Line= 3
      1447890.91       6834476.9        1448755.        6833488.
      1449088.81      6832456.08
#Sta/Elev= 30
    3683 2357.83  3692.5 2356.79  3748.5 2337.79  3840.9 2315.86  3933.6  2302.2
  4095.9 2285.37  4224.1 2277.01  4414.8 2269.07  4783.8 2264.89  4868.6 2260.64
  4931.3 2254.13  5003.4 2246.33  5003.9 2245.83  5010.1 2246.33  5101.3 2249.53
  5241.6 2250.82  5337.6 2255.86  5458.7  2266.1  5593.7 2285.45  5637.4 2297.78
  5689.7 2309.26    5753 2327.41    5816 2351.11    5855 2372.29  5924.3 2403.45
  5931.6 2408.96  5963.2 2423.58  6015.1 2442.12  6049.3 2444.89  6080.8 2446.44
#Mann= 5 ,-1 , 0
    3683     .07       0  4931.3     .16       0  5003.4     .07       0
  5010.1     .16       0  6049.3     .07       0
Bank Sta=5003.4,5010.1
XS Rating Curve= 0 ,0
Exp/Cntr=0.3,0.1

Type RM Length L Ch R = 1 ,19947   ,466,466,466
BEGIN DESCRIPTION:
WEAVER SPRINGS CREEK TRIB 1 30.0
END DESCRIPTION:
XS GIS Cut Line= 3
      1448021.13      6834549.81        1449205.        6833588.
      1449224.22      6832586.31
#Sta/Elev= 30
  3474.7 2331.45  3514.6  2321.6  3642.4 2301.74  3770.3 2288.09  3862.9 2280.97
  3912.5 2279.45  3926.9 2276.69  4232.1 2263.95  4452.7 2257.41  4516.6 2253.05
  4879.4 2248.63  4922.5 2244.33  4993.4 2242.02  4993.9 2241.52  5000.2 2242.02
  5047.2 2242.39  5420.1 2247.34  5500.1  2253.1  5600.1 2266.75  5710.2 2293.64
  5740.2  2303.7  5778.5  2312.8  5783.5 2309.86  5790.2 2312.57  5820.2 2327.94
  5870.2  2359.7  5900.2    2383  5940.2 2403.21  5998.6 2430.16  6001.9 2430.16
#Mann= 4 ,-1 , 0
  3474.7     .07       0  4993.4     .07       0  5000.2     .07       0
  5047.2     .16       0
Bank Sta=4993.4,5000.2
XS Rating Curve= 0 ,0
Exp/Cntr=0.3,0.1

Type RM Length L Ch R = 1 ,19481   ,496,496,496
BEGIN DESCRIPTION:
WEAVER SPRINGS CREEK TRIB 1 29.0
END DESCRIPTION:
XS GIS Cut Line= 3
      1448375.28      6834874.47        1449655.        6833488.
      1449302.54      6832432.37
#Sta/Elev= 30
  3131.3  2280.6  3361.9 2271.45  3673.3 2266.29  3878.6 2259.57  3984.6 2259.48
  4522.8 2249.52    4728 2239.45  4855.1 2239.16  4876.6 2235.95  4979.2 2230.85
  4979.7 2230.35    4986 2230.85  5065.5 2234.82  5160.3 2233.22  5228.9 2239.05
  5376.2 2239.97  5460.2 2243.24  5597.5 2252.52  5634.3 2257.68  5665.9 2266.19
  5823.9 2327.01  5881.9 2351.58  5924.8 2372.97  6008.3 2402.45  6019.6 2409.42
  6039.9 2413.37  6047.3  2417.9  6076.8 2430.91  6093.4  2443.8    6131 2446.25
#Mann= 6 ,-1 , 0
  3131.3     .16       0  3361.9     .07       0  4979.2     .07       0
    4986     .07       0  5460.2     .16       0  6047.3     .07       0
Bank Sta=4979.2,4986
XS Rating Curve= 0 ,0
Exp/Cntr=0.3,0.1

Type RM Length L Ch R = 1 ,18985   ,139,139,139
BEGIN DESCRIPTION:
WEAVER SPRINGS CREEK TRIB 1 28.0
END DESCRIPTION:
XS GIS Cut Line= 4
      1450182.25      6834694.07      1450093.71      6833496.13
        1449905.        6833138.      1449449.08      6832339.62
#Sta/Elev= 30
  3398.3 2276.44  3538.9 2275.77  3795.5 2270.53  3885.7 2266.87  3945.9 2262.06
    4006 2261.34  4026.1  2258.6  4375.3  2248.1  4518.3 2237.25  4675.6 2233.61
  4802.5 2231.41  4873.9 2230.94    4968 2227.54  4968.5 2227.04  4980.1 2227.54
  5039.6 2232.19  5091.1 2232.84  5291.6 2238.68  5362.9 2246.13  5545.6 2281.55
  5555.1 2280.96  5560.8 2284.59  5576.7 2286.04  5582.4 2290.27  5591.6 2291.22
    5604 2296.69  5649.2 2309.63  5700.5  2329.2  5781.2  2369.2  5923.7 2443.61
#Mann= 9 ,-1 , 0
  3398.3     .16       0  3538.9     .07       0  4675.6     .16       0
  4802.5     .07       0  4873.9     .16       0    4968     .07       0
  4980.1     .16       0  5091.1     .07       0  5362.9     .16       0
Bank Sta=4968,4980.1
XS Rating Curve= 0 ,0
Exp/Cntr=0.3,0.1

Type RM Length L Ch R = 1 ,18846   ,689,689,689
BEGIN DESCRIPTION:
WEAVER SPRINGS CREEK TRIB 1 27.0
END DESCRIPTION:
XS GIS Cut Line= 4
        1450280.      6834162.98      1450172.51      6833433.23
      1450029.95      6833087.82      1449489.25      6832264.25
#Sta/Elev= 30
  3888.7 2264.49  4232.1 2254.56  4371.5 2248.51  4469.9 2239.55  4627.7 2233.85
  4741.7 2230.92  4826.7 2232.37  4967.4 2227.12  4982.9 2222.84  4983.4 2222.34
    4995 2222.84  5017.9 2228.31  5062.7 2230.88    5256 2233.99  5328.3 2237.62
  5368.6 2242.66  5415.7 2246.76  5436.8 2251.35    5473 2263.56  5538.1 2277.19
  5638.7 2306.06    5711 2332.02  5747.2 2348.07  5813.2 2377.78  5855.7 2399.98
  5876.8 2407.97  5891.9 2419.57  5903.6 2424.88  5943.1 2442.75  5985.2 2446.57
#Mann= 7 ,-1 , 0
  3888.7     .07       0  4627.7     .16       0  4982.9     .07       0
    4995     .16       0  5062.7     .07       0  5368.6     .16       0
  5903.6     .07       0
Bank Sta=4982.9,4995
XS Rating Curve= 0 ,0
Exp/Cntr=0.3,0.1

Type RM Length L Ch R = 1 ,18157   ,621,621,621
BEGIN DESCRIPTION:
WEAVER SPRINGS CREEK TRIB 1 26.0
END DESCRIPTION:
XS GIS Cut Line= 3
      1450425.55      6834021.56        1450555.        6832738.
      1449791.89      6831894.83
#Sta/Elev= 30
  3709.7 2259.46  3813.8 2259.26  3994.7 2252.65  4135.4 2251.19  4391.8 2240.54
  4557.5 2226.89  4859.1    2225  4952.2 2218.36  4953.5 2216.38    4954 2215.88
  4965.6 2216.38  4997.3 2220.78  5323.5 2230.37  5493.1 2240.79  5601.6    2251
  5622.6 2257.96    5738 2276.45  5842.3 2282.96  5891.6  2289.6    5899 2293.43
  5962.6 2309.39  6005.1 2316.83  6047.7 2330.48  6082.9  2345.1  6090.3 2345.45
  6097.1 2351.26  6104.5 2350.82  6111.2 2356.22  6125.4 2362.25    6137 2363.85
#Mann= 7 ,-1 , 0
  3709.7     .07       0  4391.8     .16       0  4953.5     .07       0
  4965.6     .16       0  5323.5     .07       0  5493.1     .16       0
    5738     .07       0
Bank Sta=4953.5,4965.6
XS Rating Curve= 0 ,0
Exp/Cntr=0.3,0.1

Type RM Length L Ch R = 1 ,17536   ,691,691,691
BEGIN DESCRIPTION:
WEAVER SPRINGS CREEK TRIB 1 25.0
END DESCRIPTION:
XS GIS Cut Line= 3
      1450599.15      6833943.47      1451049.03      6832440.14
      1449918.86      6831466.09
#Sta/Elev= 30
  3430.8 2254.23    3440 2254.21  3746.1 2250.69  4049.6 2239.75  4386.4 2224.38
  4469.9 2219.09  4477.6 2216.43  4483.1 2218.97  4490.8 2215.79  4510.7 2218.44
  4556.5 2217.83  4699.5  2220.3  4801.6 2217.94  4960.5 2216.85  4992.4 2211.93
  4992.9 2211.43  5004.6 2211.93  5011.4 2214.25  5060.8 2218.05  5343.6 2223.56
  5500.3  2227.6    5683 2234.66    5763 2238.45  6082.2  2269.6  6145.8 2272.43
    6238 2280.29  6330.2 2291.33  6408.1 2307.93  6450.8 2320.78    6492 2337.23
#Mann= 11 ,-1 , 0
  3430.8     .16       0    3440     .07       0  4049.6     .16       0
  4483.1     .07       0  4556.5     .16       0  4801.6     .07       0
  4992.4     .07       0  5004.6     .07       0  5343.6     .16       0
  5500.3     .07       0    5683     .16       0
Bank Sta=4992.4,5004.6
XS Rating Curve= 0 ,0
Exp/Cntr=0.3,0.1

Type RM Length L Ch R = 1 ,16845   ,477,477,477
BEGIN DESCRIPTION:
WEAVER SPRINGS CREEK TRIB 1 23.0
END DESCRIPTION:
XS GIS Cut Line= 3
      1452118.26      6833538.92        1451655.        6832488.
      1450454.99      6831387.99
#Sta/Elev= 30
  3851.5 2244.42  3922.6 2245.74  4038.3  2243.3  4180.4 2233.95  4247.6 2230.56
    4271 2231.25  4317.6 2227.17  4387.6  2225.2  4453.6 2220.88  4660.5 2212.68
  4879.8  2211.8  4910.2 2210.32  4945.4 2205.83  4991.1 2208.36  4997.3 2204.34
    5007 2202.97  5007.5 2202.47  5020.7 2202.97  5028.1 2208.88  5042.2 2210.72
  5216.3 2213.43  5254.3  2213.9  5467.1 2214.21  5761.7 2219.17  5829.2 2220.98
  5919.2 2223.25  5979.5 2225.06  6186.9 2236.65  6499.1 2257.32  6627.9 2266.44
#Mann= 11 ,-1 , 0
  3851.5     .07       0    5007     .07       0  5020.7     .07       0
  5216.3     .16       0  5254.3     .07       0  5761.7     .16       0
  5829.2     .07       0  5919.2     .16       0  5979.5     .07       0
  6186.9     .16       0  6499.1     .07       0
Bank Sta=5007,5020.7
XS Rating Curve= 0 ,0
Exp/Cntr=0.3,0.1

Type RM Length L Ch R = 1 ,16368   ,1157,1157,1157
BEGIN DESCRIPTION:
WEAVER SPRINGS CREEK TRIB 1 22.0
END DESCRIPTION:
XS GIS Cut Line= 3
      1452213.75      6833417.41        1452055.        6832288.
      1450912.91      6830901.54
#Sta/Elev= 30
  3854.2 2239.97  3956.3 2238.92  4045.5 2232.72  4093.8 2227.91  4165.1 2225.11
  4170.1 2225.96  4236.3 2222.11  4455.2 2215.97  4526.4 2214.48  4560.5 2215.14
    4669 2210.01  4775.2 2208.78  4899.6 2208.03  4959.1 2206.31  4974.5 2201.83
  4977.8 2199.43  4978.3 2198.93  4991.5 2199.43  5030.6 2205.74  5080.1 2207.19
  5719.9 2210.55  5804.6  2212.7    5876 2216.58  5940.1 2220.62  6088.6  2226.6
  6259.4    2237  6273.7 2239.05  6529.1 2258.28  6664.6  2270.8    6791  2286.4
#Mann= 7 ,-1 , 0
  3854.2     .07       0  4775.2     .16       0  4899.6     .07       0
  4977.8     .07       0  4991.5     .07       0    5876     .16       0
  6088.6     .07       0
Bank Sta=4977.8,4991.5
XS Rating Curve= 0 ,0
Exp/Cntr=0.3,0.1

Type RM Length L Ch R = 1 ,15211   ,1971,1971,1971
BEGIN DESCRIPTION:
WEAVER SPRINGS CREEK TRIB 1 21.0
END DESCRIPTION:
XS GIS Cut Line= 3
      1453562.41      6833250.13      1453070.68      6832254.52
       1451349.8      6830703.23
#Sta/Elev= 30
  3903.3 2261.23  4381.3 2230.94  4605.8 2221.49    4920 2212.67  4942.4 2208.69
  4970.5 2207.09  4987.3 2202.02  5001.7 2192.57  5002.2 2192.07  5016.4 2192.57
  5036.3  2197.3  5156.6 2198.31  5199.2 2201.44  5765.7 2198.66  6056.4 2200.63
    6155 2198.68  6233.1 2201.92  6424.1  2205.1  6568.4 2209.85  6658.2 2215.28
  6835.1 2225.34  6898.7 2231.31  7026.5 2238.56  7054.3 2241.23  7075.8 2245.27
  7125.1 2247.25  7139.3 2249.58    7217 2255.22  7281.3 2262.83  7330.6 2266.37
#Mann= 5 ,-1 , 0
  3903.3     .07       0  5001.7     .07       0  5016.4     .07       0
  6568.4     .16       0  6658.2     .07       0
Bank Sta=5001.7,5016.4
XS Rating Curve= 0 ,0
Exp/Cntr=0.3,0.1

Type RM Length L Ch R = 1 ,13240   ,862,862,862
BEGIN DESCRIPTION:
WEAVER SPRINGS CREEK TRIB 1 20.0
END DESCRIPTION:
XS GIS Cut Line= 3
      1453904.99      6832037.99        1452705.        6830838.
      1451353.24      6830525.75
#Sta/Elev= 30
  3298.7 2231.09  3510.8 2218.79  4019.9 2197.06  4203.8 2193.85    4458 2192.59
  4552.1 2191.55    4727 2190.12  4939.2 2186.01    4986 2183.06    5006 2182.26
    5019  2178.3  5019.5  2177.8    5034  2178.3  5038.4 2181.35  5067.6 2185.47
  5159.5 2193.95  5417.6  2207.3    5745 2223.63  5765.5 2226.46  5995.9 2239.36
  6104.2 2249.09  6129.3 2249.51    6172  2254.4  6196.6 2255.81  6219.9 2254.67
  6247.9 2255.68  6262.6 2258.93  6268.4 2262.18  6288.9 2266.56  6383.1 2280.17
#Mann= 9 ,-1 , 0
  3298.7     .07       0    4458     .16       0  4552.1     .07       0
    4986     .16       0    5019     .07       0    5034     .16       0
  5038.4     .07       0  5159.5     .16       0  5417.6     .07       0
Bank Sta=5019,5034
XS Rating Curve= 0 ,0
Exp/Cntr=0.3,0.1

Type RM Length L Ch R = 1 ,12378   ,883,883,883
BEGIN DESCRIPTION:
Mapping XS 91f88f4e
END DESCRIPTION:
XS GIS Cut Line= 3
      1453817.64      6831568.46      1453293.32      6830651.77
      1452091.92      6830353.16
#Sta/Elev= 30
  3942.8 2207.07  3959.4 2207.73  3975.2 2205.12  4150.7 2198.52  4238.6 2192.17
  4276.1 2193.34  4507.8 2187.18  4684.8 2185.56  4802.9 2182.35  4926.6  2182.6
  4948.2 2179.44  4969.8  2174.4  4972.3  2172.4  4972.8  2171.9  4987.4  2172.4
  4991.7 2175.89  4998.1  2176.7  5062.8 2179.01  5204.7 2187.35  5333.2 2190.24
    5356 2190.52  5388.7 2190.79  5434.9 2186.91  5488.9 2189.34  5512.3 2192.02
  5584.5  2191.2  5742.3 2201.91  5835.4 2204.55  5990.1 2210.17  6236.8 2222.67
#Mann= 9 ,-1 , 0
  3942.8     .07       0  4972.3     .07       0  4987.4     .07       0
  5062.8     .16       0  5333.2     .07       0    5356     .16       0
  5434.9     .07       0  5742.3     .16       0  5835.4     .07       0
Bank Sta=4972.3,4987.4
XS Rating Curve= 0 ,0
Exp/Cntr=0.3,0.1

Type RM Length L Ch R = 1 ,11495   ,125,125,125
BEGIN DESCRIPTION:
WEAVER SPRINGS CREEK TRIB 1 19.0
END DESCRIPTION:
XS GIS Cut Line= 5
      1454755.12      6831148.28       1454215.2      6830246.39
      1453885.34      6830194.31       1453568.5      6830302.81
      1452275.05       6830354.9
#Sta/Elev= 30
  3477.1 2213.35  3660.2 2205.23  3893.5 2199.26  4132.7  2196.9  4344.7 2191.94
  4609.2 2181.53  4681.8 2176.81  4894.3 2177.08  4946.3 2171.35  4957.7 2168.65
  4982.9 2166.88  5008.9 2168.54  5014.2 2166.65  5031.7 2167.44  5037.8  2166.1
  5038.3  2165.6  5053.1  2166.1  5116.2 2175.02    5148 2177.08  5310.7 2182.85
  5511.1 2186.23  5593.6 2186.85  5702.4 2188.75  5851.1 2186.43  5911.2 2189.34
  5961.2 2189.31  6041.3  2198.4  6227.7 2204.34  6236.5 2204.45  6491.6 2212.81
#Mann= 7 ,-1 , 0
  3477.1     .07       0  5037.8     .07       0  5053.1     .07       0
  5511.1     .16       0  5593.6     .07       0  6227.7     .16       0
  6236.5     .07       0
Bank Sta=5037.8,5053.1
XS Rating Curve= 0 ,0
Exp/Cntr=0.3,0.1

Type RM Length L Ch R = 1 ,11370   ,565,565,565
BEGIN DESCRIPTION:
WEAVER SPRINGS CREEK TRIB 1 18.0
END DESCRIPTION:
XS GIS Cut Line= 6
      1454848.39      6831209.21      1454226.05      6830102.73
      1453835.42      6830076.68      1453703.05      6830133.11
      1453492.54      6830224.25      1452200.43       6830229.9
#Sta/Elev= 30
  3192.8 2216.32  3291.6 2213.45  3410.2  2206.2  3534.5 2201.58  3723.8 2197.94
  3739.7 2196.42  3966.6 2193.59  4004.3 2191.32  4112.6 2191.16  4349.7 2186.16
  4458.1  2183.2  4623.7 2174.68    4876 2175.76  4975.6 2170.04  4984.7  2168.3
  4986.1 2166.25  4986.6 2165.75  5001.4 2166.25  5022.7 2170.92  5069.7 2171.32
  5122.1 2176.11  5225.5 2180.95  5306.4 2181.74  5523.4 2184.55  5714.6 2184.33
  5804.6 2190.46  5984.6 2194.99  6074.6 2200.27  6374.6 2209.44  6519.2 2215.93
#Mann= 5 ,-1 , 0
  3192.8     .07       0  4986.1     .07       0  5001.4     .07       0
  5306.4     .16       0  5523.4     .07       0
Bank Sta=4986.1,5001.4
XS Rating Curve= 0 ,0
Exp/Cntr=0.3,0.1

Type RM Length L Ch R = 1 ,10805   ,550,550,550
BEGIN DESCRIPTION:
WEAVER SPRINGS CREEK TRIB 1 17.0
END DESCRIPTION:
XS GIS Cut Line= 3
      1454354.98      6829937.99      1453808.97      6829639.65
      1453054.14      6829369.84
#Sta/Elev= 30
  4377.8 2186.39  4407.7 2184.24  4445.6 2183.12  4480.3 2180.47  4573.8  2176.1
  4696.1 2171.36  4735.5 2170.55  4822.2 2170.34  4834.3 2170.07    4865  2169.5
  4886.8 2167.72  4914.3 2166.66  4990.2 2166.85  4991.1 2161.01  4991.6 2160.51
  5007.2 2160.51  5007.7 2161.01  5014.6 2161.38  5019.9 2163.46  5025.5 2167.11
  5050.7 2174.71  5076.2 2177.15  5137.8 2179.23    5194 2179.65  5386.9  2183.8
  5409.5 2183.91  5418.4 2184.95  5425.6 2184.91  5630.8 2191.47  5801.6  2198.9
#Mann= 9 ,-1 , 0
  4377.8     .07       0  4573.8     .16       0  4735.5     .07       0
  4822.2     .16       0  4834.3     .07       0  4991.1     .07       0
  5007.7     .07       0  5386.9     .16       0  5425.6     .07       0
Bank Sta=4991.1,5007.7
XS Rating Curve= 0 ,0
Exp/Cntr=0.3,0.1

Type RM Length L Ch R = 1 ,10255   ,305,305,305
BEGIN DESCRIPTION:
WEAVER SPRINGS CREEK TRIB 1 16.0
END DESCRIPTION:
XS GIS Cut Line= 3
      1454422.19      6829852.47      1454232.13      6829349.09
      1453700.18      6828772.85
#Sta/Elev= 30
    4448 2184.16  4495.5 2184.53  4559.7 2183.28  4626.6 2180.37  4721.1 2173.07
  4760.3 2170.73  4907.1 2162.65  4944.5 2161.67  4953.8  2157.5  4954.3    2157
  4970.4  2157.5    4984  2162.5  4991.8 2162.84  4999.2 2164.98  5020.1 2166.96
    5112 2170.04  5367.2 2172.48  5437.5 2176.54  5494.2  2178.6  5544.1 2182.13
  5614.4 2184.93  5650.1 2188.06  5656.9 2187.83  5664.3 2189.27  5671.1 2189.23
  5692.6 2192.05  5699.5 2191.77  5713.6 2192.97    5721 2194.27  5770.3 2196.98
#Mann= 5 ,-1 , 0
    4448     .07       0  4721.1     .16       0  4760.3     .07       0
  4953.8     .07       0  4970.4     .07       0
Bank Sta=4953.8,4970.4
XS Rating Curve= 0 ,0
Exp/Cntr=0.3,0.1

Type RM Length L Ch R = 1 ,9950    ,431,431,431
BEGIN DESCRIPTION:
WEAVER SPRINGS CREEK TRIB 1 15.0
END DESCRIPTION:
XS GIS Cut Line= 4
      1454467.91      6829843.14      1454561.66       6829280.6
      1454392.39      6829132.17      1454405.41      6828546.24
#Sta/Elev= 30
    4324 2183.36    4390 2183.74  4511.7  2180.1  4542.1 2178.59  4613.1 2172.39
  4633.3  2171.6  4639.6 2170.42  4836.1  2167.7    4922 2164.53  4936.3 2161.78
  4943.1 2162.19  4957.2 2160.06  4964.7 2158.36  4970.7 2155.05  4971.2 2154.55
  4987.3 2155.05  4993.2 2159.88  5007.4 2161.21  5163.6 2161.69  5208.1 2160.62
  5243.6 2159.97  5253.6 2161.24  5263.6 2160.96  5273.6 2162.05  5293.6 2166.24
  5363.7 2172.25  5403.9 2177.41  5501.8 2183.26  5567.4 2186.09  5705.5 2193.14
#Mann= 7 ,-1 , 0
    4324     .07       0  4970.7     .07       0  4987.3     .07       0
  5208.1     .16       0  5403.9     .07       0  5501.8     .16       0
  5567.4     .07       0
Bank Sta=4970.7,4987.3
XS Rating Curve= 0 ,0
Exp/Cntr=0.3,0.1

Type RM Length L Ch R = 1 ,9519    ,278,278,278
BEGIN DESCRIPTION:
WEAVER SPRINGS CREEK TRIB 1 14.0
END DESCRIPTION:
XS GIS Cut Line= 3
        1454605.      6829737.98       1454767.3      6828937.67
        1454658.      6828535.77
#Sta/Elev= 30
  4183.4 2181.27  4244.6 2180.44  4275.2 2179.11    4310 2176.29  4346.6 2171.88
  4387.5    2169  4469.1 2167.47  4664.7 2166.58  4754.8  2164.9  4785.4 2163.35
  4811.6  2160.7  4979.3 2158.42  4989.5 2157.66    5000 2155.59  5001.6 2154.59
  5002.1 2154.09  5018.5 2154.59  5021.7 2155.77  5044.2 2161.73  5051.5 2163.82
  5061.3 2168.14  5066.5 2168.67  5072.2  2174.9  5082.6 2180.75  5113.7 2182.43
  5134.4 2182.29  5206.9 2188.99    5238 2193.66  5260.2 2195.31  5416.5 2197.98
#Mann= 5 ,-1 , 0
  4183.4     .07       0  5001.6     .07       0  5018.5     .07       0
  5021.7     .16       0  5044.2     .07       0
Bank Sta=5001.6,5018.5
XS Rating Curve= 0 ,0
Exp/Cntr=0.3,0.1

Type RM Length L Ch R = 1 ,9241    ,376,376,376
BEGIN DESCRIPTION:
Mapping XS 1b87f6dd
END DESCRIPTION:
XS GIS Cut Line= 3
      1454764.78      6829690.55      1455046.04      6828937.99
      1454772.58      6828588.96
#Sta/Elev= 30
  4196.6 2175.13  4252.7  2169.9  4384.5    2165  4402.2 2165.78  4666.1 2164.34
  4850.5 2160.81  4897.8 2158.25  4903.9 2156.54  4914.6 2155.85    4978 2155.95
  4980.9 2151.44  4981.4 2150.94  4997.8 2151.44  5003.2 2152.09  5008.1 2154.12
  5022.5 2155.68  5142.8 2159.01  5279.3 2167.81  5300.1 2171.06  5306.4 2173.96
  5320.9 2176.23  5349.8 2177.36  5385.1 2183.72  5393.2 2183.93  5399.5 2187.12
    5414 2187.68  5420.4 2190.45  5428.5 2189.91  5434.8 2191.51  5443.4 2190.29
#Mann= 3 ,-1 , 0
  4196.6     .07       0  4980.9     .07       0  4997.8     .07       0
Bank Sta=4980.9,4997.8
XS Rating Curve= 0 ,0
Exp/Cntr=0.3,0.1

Type RM Length L Ch R = 1 ,8865    ,833,833,833
BEGIN DESCRIPTION:
Mapping XS 7f3bdc6a
END DESCRIPTION:
XS GIS Cut Line= 4
      1454963.14      6829672.81      1455395.02      6829093.35
      1455434.09      6828854.64      1454934.93       6828448.8
#Sta/Elev= 30
  4133.9 2165.41    4175 2165.37  4339.4    2162  4381.4  2162.4  4575.3 2161.24
  4810.9 2157.74  4872.2 2155.99  4948.7  2151.8  5003.9 2153.64  5015.2 2150.15
  5015.6  2148.9  5016.1  2148.4  5032.6  2148.9  5034.3 2151.69  5044.4 2153.08
  5071.5 2155.61  5098.5 2156.95  5102.4 2158.31  5110.2  2158.7  5358.1 2159.28
  5436.4 2160.02  5471.6 2161.17  5522.6 2160.71  5549.9 2161.37  5586.5 2163.53
  5642.5 2164.22  5677.7 2165.85    5700 2167.82  5735.2 2167.74  5741.8 2168.63
#Mann= 3 ,-1 , 0
  4133.9     .07       0  5015.6     .07       0  5032.6     .07       0
Bank Sta=5015.6,5032.6
XS Rating Curve= 0 ,0
Exp/Cntr=0.3,0.1

Type RM Length L Ch R = 1 ,8032    ,450,450,450
BEGIN DESCRIPTION:
Mapping XS e25ed4b3
END DESCRIPTION:
XS GIS Cut Line= 4
      1456022.19      6829776.53      1456162.82      6829227.03
      1456071.67      6828911.93      1455329.76      6828386.08
#Sta/Elev= 30
  4444.5 2167.62  4477.6 2167.46  4484.3 2166.43  4513.2 2165.08  4628.8 2161.96
  4635.6 2161.06  4676.5 2159.19  4798.9 2156.72  4855.9 2154.53  4866.2 2155.17
  4938.5 2149.82  4990.1  2149.3  5002.9  2148.5  5008.6 2147.32  5010.3 2144.71
  5010.8 2144.21  5027.5 2144.71  5031.5 2147.08  5041.9 2148.38  5130.1 2147.93
  5168.9 2149.73  5177.3 2150.96  5236.1  2152.4  5260.5  2151.2  5390.3 2150.83
  5519.5 2152.59  5547.8 2153.58  5654.8 2154.06  5785.3 2156.22  6249.1 2156.26
#Mann= 3 ,-1 , 0
  4444.5     .07       0  5010.3     .07       0  5027.5     .07       0
Bank Sta=5010.3,5027.5
XS Rating Curve= 0 ,0
Exp/Cntr=0.3,0.1

Type RM Length L Ch R = 1 ,7582    ,599,599,599
BEGIN DESCRIPTION:
Mapping XS 7fe559d7
END DESCRIPTION:
XS GIS Cut Line= 3
      1456544.76      6829962.29      1456569.07        6829122.
      1455492.66      6828417.13
#Sta/Elev= 30
    4161 2171.27  4205.3 2170.79  4235.3 2169.19  4375.4 2165.45  4455.4 2161.99
  4505.4 2160.99  4555.5 2158.68  4565.5 2158.93  4585.5 2157.46  4655.5 2155.48
  4675.5 2153.93  4684.2 2155.15  4692.9 2154.72  4783.1 2152.99  4815.6 2153.33
  4935.6 2148.89  4955.6 2146.99  4975.6 2143.85    4977 2141.58  4977.5 2141.08
  4994.3 2141.58  5001.1 2144.62  5086.7 2145.09  5200.9 2148.68  5440.4 2149.44
  5512.7  2150.1  5527.8  2151.1  5606.2 2150.79  5744.9  2153.5  6288.3 2155.61
#Mann= 7 ,-1 , 0
    4161     .07       0  4692.9     .16       0  4783.1     .07       0
    4977     .07       0  4994.3     .07       0  5086.7    .035       0
  5200.9     .07       0
Bank Sta=4977,4994.3
XS Rating Curve= 0 ,0
Exp/Cntr=0.3,0.1

Type RM Length L Ch R = 1 ,6983    ,536,536,536
BEGIN DESCRIPTION:
Mapping XS d0d2b6c0
END DESCRIPTION:
XS GIS Cut Line= 3
      1457822.57      6829403.27      1456957.96      6828701.86
      1455544.81      6828316.45
#Sta/Elev= 30
  3885.1  2165.3  3958.8 2165.25    4039 2163.28    4221 2161.42  4520.9 2161.34
  4612.6  2160.5  4668.6  2158.3  4699.5 2158.73  4868.3 2152.02  4897.1 2148.58
  4917.9 2147.55  4953.1 2142.88  4967.5 2140.35  4973.1  2137.3  4973.6  2136.8
  4990.6  2137.3  4996.2 2140.42  5011.9 2141.24    5043 2140.23  5097.4 2142.59
  5115.5 2143.16  5136.3 2141.46  5167.3 2141.43  5278.1  2144.7  5297.5 2145.87
    5491  2145.7  5739.9 2148.17  5911.9 2149.57  6358.2  2153.8  6463.2 2153.65
#Mann= 10 ,-1 , 0
  3885.1     .07       0    4039    .045       0  4520.9    .035       0
  4699.5     .07       0  4973.1     .07       0  4990.6     .07       0
  5097.4    .035       0  5278.1     .07       0  5739.9    .035       0
  5911.9     .07       0
Bank Sta=4973.1,4990.6
XS Rating Curve= 0 ,0
Exp/Cntr=0.3,0.1

Type RM Length L Ch R = 1 ,6447    ,192,192,192
BEGIN DESCRIPTION:
Mapping XS 70107cef
END DESCRIPTION:
XS GIS Cut Line= 3
      1457666.27      6828462.27      1456947.54      6828312.97
      1455454.53       6828035.2
#Sta/Elev= 30
  4294.1  2156.1  4350.4 2156.15  4404.3 2156.29  4662.6 2155.89  4736.4 2153.27
  4781.4 2149.88  4881.6 2145.41  4938.8 2140.81  5000.1 2138.58  5020.6 2137.13
  5023.3 2134.72  5023.8 2134.22  5040.8 2134.72  5071.4 2137.65  5079.6 2136.02
  5084.7 2139.03  5091.8 2137.39    5102 2137.84  5112.1  2140.1  5122.3 2140.73
  5137.5 2140.23  5631.2 2144.06  5703.5 2144.55  5773.3 2144.96  5824.1 2146.48
  6012.2 2146.85  6098.8 2148.43  6363.2 2149.97  6403.9 2151.26  6546.8 2151.77
#Mann= 8 ,-1 , 0
  4294.1    .035       0  4350.4     .07       0  4404.3    .035       0
  4662.6     .07       0  5023.3     .07       0  5040.8     .07       0
  5631.2    .035       0  5703.5     .07       0
Bank Sta=5023.3,5040.8
XS Rating Curve= 0 ,0
Exp/Cntr=0.3,0.1

Type RM Length L Ch R = 1 ,6255    ,811,811,811
BEGIN DESCRIPTION:
Mapping XS 85909b21
END DESCRIPTION:
XS GIS Cut Line= 3
      1457558.63      6828285.19      1456951.01      6828153.25
      1455430.21      6827868.53
#Sta/Elev= 30
  4382.3 2156.16  4549.7 2155.74  4600.9 2154.84  4662.3 2152.03  4676.5 2152.19
  4769.7 2147.69  4887.4 2145.97  4906.9 2143.33    4912 2144.03  4938.6 2140.76
    4956 2135.85  4961.1 2136.68  4970.7 2133.56  4971.2 2133.06  4988.3 2133.56
  4989.8 2136.15  4999.5 2137.02  5091.6 2139.03  5336.2 2138.93    5494 2141.05
  5691.8  2142.3  5709.5 2143.11  5714.6 2142.54  5722.4 2143.32  5885.1  2145.5
  5905.5 2144.97  6040.4 2145.72  6190.3 2147.82  6255.9 2147.86  6551.3 2151.83
#Mann= 3 ,-1 , 0
  4382.3     .07       0  4970.7     .07       0  4988.3     .07       0
Bank Sta=4970.7,4988.3
XS Rating Curve= 0 ,0
Exp/Cntr=0.3,0.1

Type RM Length L Ch R = 1 ,5444    ,473,473,473
BEGIN DESCRIPTION:
WEAVER SPRINGS CREEK TRIB 1 10.0
END DESCRIPTION:
XS GIS Cut Line= 3
      1457454.99        6827788.        1456455.        6827588.
      1455555.05      6827787.99
#Sta/Elev= 30
  3980.7 2153.84  4052.1  2154.2  4143.9 2151.74  4225.4 2145.69    4256 2144.96
  4276.4 2143.67  4419.2 2142.46  4684.4 2142.34  4857.7 2135.94  4990.3 2132.24
  4997.9 2130.01  5000.5 2130.01  5001.9 2128.09  5002.4 2127.59    5019 2127.59
  5019.5 2128.09  5019.7 2130.18  5024.8 2132.15  5073.5 2135.41  5204.1 2134.98
  5225.9 2136.09  5246.3 2138.03  5369.3 2138.32  5430.7 2140.94  5522.9 2143.64
  5543.4  2145.3  5635.6  2147.2  5799.5 2148.71    5861 2150.51  5922.4  2151.1
#Mann= 3 ,-1 , 0
  3980.7     .07       0  5001.9     .07       0  5019.5     .07       0
Bank Sta=5001.9,5019.5
XS Rating Curve= 0 ,0
Exp/Cntr=0.3,0.1

Type RM Length L Ch R = 1 ,4971    ,746,746,746
BEGIN DESCRIPTION:
WEAVER SPRINGS CREEK TRIB 1 9.0
END DESCRIPTION:
XS GIS Cut Line= 3
      1457354.99      6827687.99        1456355.        6827188.
      1455730.04      6826913.02
#Sta/Elev= 30
  3877.4 2152.82  3944.5  2149.7  3975.2 2146.83  4056.3 2143.59  4070.2 2144.12
  4078.6  2143.1  4190.4 2141.39  4450.4 2140.15  4637.7  2137.4  4771.8 2133.67
  4869.6 2132.22  4897.6  2132.4    4906 2131.66  4973.1 2130.27  4981.4 2129.16
  4983.8 2125.57  4984.3 2125.07    5001 2125.07  5001.5 2125.57  5004.4 2128.32
  5009.8 2129.86  5033.2  2130.8  5056.5  2133.4  5079.8 2134.44    5202 2135.14
  5312.3 2134.77  5358.4 2135.18  5428.5 2136.91  5457.3 2136.68  5678.2  2139.2
#Mann= 3 ,-1 , 0
  3877.4     .07       0  4983.8     .07       0  5001.5     .07       0
Bank Sta=4983.8,5001.5
XS Rating Curve= 0 ,0
Exp/Cntr=0.3,0.1
