--- Noodle Creek.prj (project) ---

Proj Title=Noodle Creek Base Level Engineering
Current Plan=p01
Default Exp/Contr=0.3,0.1
English Units
Geom File=g01
Flow File=f01
Plan File=p01
Y Axis Title=Elevation
X Axis Title(PF)=Main Channel Distance
X Axis Title(XS)=Station
BEGIN DESCRIPTION:
Noodle Creek
END DESCRIPTION:
DSS Export Rating Curves= 0
DSS Export Rating Curve Sorted= 0
DSS Export Volume Flow Curves= 0
DXF OffsetX= 0
DXF OffsetY= 0
DXF ScaleX= 1
DXF ScaleY= 10

--- Noodle Creek.p01 (plan) ---

Plan Title=Multiple Run
Short Identifier=Multiple
Geom File=g01
Flow File=f01
Subcritical Flow
K Sum by GR= 0
Std Step Tol= 0.01
Critical Tol= 0.01
Num of Std Step Trials= 20
Max Error Tol= 0.3
Flow Tol Ratio= 0.001
Split Flow NTrial= 30
Split Flow Tol= 0.02
Split Flow Ratio= 0.02
Log Output Level= 0
Friction Slope Method= 1
Unsteady Friction Slope Method= 2
Unsteady Bridges Friction Slope Method= 1
Parabolic Critical Depth
Global Vel Dist=  1 , 1 , 1
Global Log Level= 0
CheckData=True
Encroach Param= -1, 0, 0, 0
BEGIN DESCRIPTION:
Multiple Run
END DESCRIPTION:

--- Noodle Creek.f01 (steady flow) ---

Flow Title=Multiple
Program Version=4.10
Number of Profiles= 7
Profile Names=10-year,25-year,50-year,1pct_min,100-year,1pct_plu,500-year
River Rch & RM=Noodle Creek,Reach-1         ,171766
     531     787    1012     647    1291    2576    2130
River Rch & RM=Noodle Creek,Reach-1         ,161308
     616     915    1177     752    1501    2995    2474
River Rch & RM=Noodle Creek,Reach-1         ,155670
     672     988    1265     803    1602    3197    2605
River Rch & RM=Noodle Creek,Reach-1         ,146743
     974    1445    1857    1183    2360    4708    3859
River Rch & RM=Noodle Creek,Reach-1         ,140602
    2198    3343    4374    2828    5643   11259    9511
River Rch & RM=Noodle Creek,Reach-1         ,131780
    2198    3343    4374    2828    5643   11259    9511
River Rch & RM=Noodle Creek,Reach-1         ,128889
    2198    3343    4374    2828    5643   11259    9511
River Rch & RM=Noodle Creek,Reach-1         ,123451
    2198    3343    4374    2828    5643   11259    9511
River Rch & RM=Noodle Creek,Reach-1         ,121501
    2200    3334    4351    2806    5598   11170    9384
River Rch & RM=Noodle Creek,Reach-1         ,119091
    2200    3334    4351    2806    5598   11170    9384
River Rch & RM=Noodle Creek,Reach-1         ,116742
    2308    3496    4561    2939    5865   11701    9818
River Rch & RM=Noodle Creek,Reach-1         ,111608
    2308    3496    4561    2939    5865   11701    9818
River Rch & RM=Noodle Creek,Reach-1         ,108762
    2265    3419    4449    2860    5705   11384    9501
River Rch & RM=Noodle Creek,Reach-1         ,103396
    3072    4662    6089    3925    7832   15627   13116
River Rch & RM=Noodle Creek,Reach-1         ,99604
    3072    4662    6089    3925    7832   15627   13116
River Rch & RM=Noodle Creek,Reach-1         ,89484
    3045    4612    6014    3871    7724   15411   12896
River Rch & RM=Noodle Creek,Reach-1         ,84844
    2995    4525    5890    3784    7551   15066   12560
River Rch & RM=Noodle Creek,Reach-1         ,80082
    3099    4676    6083    3904    7790   15543   12933
River Rch & RM=Noodle Creek,Reach-1         ,78120
    3099    4676    6083    3904    7790   15543   12933
River Rch & RM=Noodle Creek,Reach-1         ,74021
    3160    4763    6191    3971    7922   15807   13130
River Rch & RM=Noodle Creek,Reach-1         ,68361
    3185    4800    6239    4001    7983   15929   13228
River Rch & RM=Noodle Creek,Reach-1         ,65857
    3163    4758    6177    3956    7893   15748   13044
River Rch & RM=Noodle Creek,Reach-1         ,59909
    3166    4759    6176    3953    7888   15738   13023
River Rch & RM=Noodle Creek,Reach-1         ,54204
    3153    4734    6137    3925    7832   15626   12906
River Rch & RM=Noodle Creek,Reach-1         ,53118
    3136    4701    6088    3890    7761   15485   12761
River Rch & RM=Noodle Creek,Reach-1         ,45319
    3125    4682    6062    3871    7723   15410   12689
River Rch & RM=Noodle Creek,Reach-1         ,42726
    3309    4961    6425    4105    8190   16340   13463
River Rch & RM=Noodle Creek,Reach-1         ,41834
    3309    4961    6425    4105    8190   16340   13463
River Rch & RM=Noodle Creek,Reach-1         ,36147
    3335    5001    6477    4137    8255   16472   13571
River Rch & RM=Noodle Creek,Reach-1         ,34917
    3329    4988    6458    4124    8228   16416   13513
River Rch & RM=Noodle Creek,Reach-1         ,29263
    3567    5325    6879    4382    8744   17446   14288
River Rch & RM=Noodle Creek,Reach-1         ,19054
    3576    5335    6890    4388    8754   17467   14294
River Rch & RM=Noodle Creek,Reach-1         ,13981
    3726    5563    7187    4579    9137   18230   14930
River Rch & RM=Noodle Creek,Reach-1         ,9100
    3721    5551    7168    4564    9106   18170   14861
River Rch & RM=Noodle Creek,Reach-1         ,5281
    3737    5573    7195    4580    9139   18235   14909
Boundary for River Rch & Prof#=Noodle Creek,Reach-1         , 1
Up Type= 0
Dn Type= 3
Dn Slope=0.001
Boundary for River Rch & Prof#=Noodle Creek,Reach-1         , 2
Up Type= 0
Dn Type= 3
Dn Slope=0.001
Boundary for River Rch & Prof#=Noodle Creek,Reach-1         , 3
Up Type= 0
Dn Type= 3
Dn Slope=0.001
Boundary for River Rch & Prof#=Noodle Creek,Reach-1         , 4
Up Type= 0
Dn Type= 3
Dn Slope=0.001
Boundary for River Rch & Prof#=Noodle Creek,Reach-1         , 5
Up Type= 0
Dn Type= 3
Dn Slope=0.001
Boundary for River Rch & Prof#=Noodle Creek,Reach-1         , 6
Up Type= 0
Dn Type= 3
Dn Slope=0.001
Boundary for River Rch & Prof#=Noodle Creek,Reach-1         , 7
Up Type= 0
Dn Type= 3
Dn Slope=0.001
DSS Import GetInterval= 0
DSS Import GetPeak= 0
DSS Import FillOption= 0

--- Noodle Creek.g01 (geometry) ---

Geom Title=Existing Conditions
Program Version=4.10

River Reach=Noodle Creek    ,Reach-1
Reach XY= 30
        1444305.        6849388.      1445510.83       6853740.3
       1448131.6      6857015.56      1455396.69      6859390.97
      1457302.29      6862182.72        1469255.        6863038.
      1470158.06       6868279.7      1472548.83      6871330.14
        1475955.        6872338.      1475660.47      6875540.45
      1478499.63      6878485.62      1477405.55      6878877.36
      1479101.87      6879889.61      1479165.75      6882497.68
      1481501.55      6883389.25      1480105.06      6885358.03
      1481747.93      6890837.99        1480605.        6893238.
      1484918.36      6899601.35      1486602.93      6900093.86
      1486305.32      6906772.98       1487355.2      6908763.08
      1486210.82      6911140.32      1487506.48      6912984.55
      1491961.21       6913095.8      1493556.56      6916484.58
      1495461.21      6915595.81      1496648.32      6918629.06
      1498849.38      6917943.62        1504455.        6925638.

Type RM Length L Ch R = 1 ,171766  ,210,210,210
BEGIN DESCRIPTION:
Noodle Creek 112.0
END DESCRIPTION:
XS GIS Cut Line= 3
      1443421.23      6849485.47      1444413.46      6849495.89
      1445280.34      6849376.14
#Sta/Elev= 30
  4056.7 2182.81  4208.2 2178.74  4234.2 2177.68  4400.5 2173.44  4524.4 2164.79
  4600.5 2154.26  4710.5 2152.66  4740.5 2141.76  4750.5 2140.91  4790.5  2141.3
  4830.5 2136.66  4850.5 2141.66  4860.5 2146.83  4890.5 2149.63  4930.5 2149.37
  4970.5 2136.69  4997.9 2135.94  4998.2 2135.44  5002.1 2135.94  5058.6 2139.34
  5067.9 2137.43  5080.8 2138.21  5131.3 2146.81  5139.8 2150.67  5144.8 2148.95
  5161.6 2152.47  5226.3 2153.04    5636 2160.06  5837.9 2168.89  5924.1 2174.77
#Mann= 8 ,-1 , 0
  4056.7     .07       0  4208.2     .16       0  4234.2     .07       0
  4524.4     .16       0  4997.9     .07       0  5002.1     .16       0
  5058.6     .07       0  5226.3     .16       0
Bank Sta=4997.9,5002.1
XS Rating Curve= 0 ,0
Exp/Cntr=0.3,0.1

Type RM Length L Ch R = 1 ,171556  ,248,248,248
BEGIN DESCRIPTION:
Mapping XS 91f2ec69
END DESCRIPTION:
XS GIS Cut Line= 4
      1443468.11      6849618.28      1444061.89      6849706.82
      1444936.89      6849667.76      1445257.24      6849568.79
#Sta/Elev= 30
  4056.1 2178.86  4283.5 2172.49  4383.1 2170.31  4450.3 2167.85  4548.4 2152.17
    4609 2149.41  4729.6 2148.23  4743.4 2146.56  4752.6 2142.36  4769.7 2137.45
  4791.2 2135.52  4809.7 2135.59  4849.7 2147.17  4939.8 2146.94  4965.6 2143.59
  4970.6 2145.19  4979.9 2143.22  4989.9 2140.27  4997.9 2133.36  4998.2 2132.86
  5002.1 2133.36  5019.9 2133.36  5029.9  2138.8  5049.9 2143.95    5080 2148.13
  5097.5 2148.33  5178.1 2148.86  5532.3 2153.55  5806.6 2165.12  5867.6 2168.25
#Mann= 11 ,-1 , 0
  4056.1     .07       0  4283.5     .16       0  4383.1     .07       0
  4450.3     .16       0  4752.6     .07       0  4791.2     .16       0
  4997.9     .07       0  5002.1     .16       0  5097.5     .07       0
  5178.1     .16       0  5806.6     .07       0
Bank Sta=4997.9,5002.1
XS Rating Curve= 0 ,0
Exp/Cntr=0.3,0.1

Type RM Length L Ch R = 1 ,171308  ,312,312,312
BEGIN DESCRIPTION:
Mapping XS ee8ceca7
END DESCRIPTION:
XS GIS Cut Line= 4
      1443489.01      6849857.87      1443996.79      6849938.59
      1444874.39      6849899.53      1445377.81      6849702.32
#Sta/Elev= 30
  4126.9 2174.01  4264.6 2170.48  4283.4  2168.9  4288.4 2167.42  4325.4 2165.95
  4354.1 2162.23    4457 2156.04  4475.1 2156.62  4487.4 2154.24  4558.2 2148.65
  4719.3  2145.3  4859.5 2144.33  4869.5 2142.61  4879.5 2138.47  4909.5 2133.61
  4929.6 2132.13  4969.6 2133.27  4997.9 2130.74  4998.2 2130.24  5002.2 2130.74
  5029.7  2131.1  5072.2 2143.24  5129.8  2144.3  5221.4 2143.47    5380    2144
  5522.5 2146.92  5638.3 2150.81  5841.6 2161.73  6041.9 2172.72  6060.2 2173.75
#Mann= 8 ,-1 , 0
  4126.9     .07       0  4354.1     .16       0  4997.9     .07       0
  5002.2     .16       0  5072.2     .07       0  5221.4     .16       0
  5841.6     .07       0  6041.9     .16       0
Bank Sta=4997.9,5002.2
XS Rating Curve= 0 ,0
Exp/Cntr=0.3,0.1

Type RM Length L Ch R = 1 ,170996  ,303,303,303
BEGIN DESCRIPTION:
Mapping XS 242d3412
END DESCRIPTION:
XS GIS Cut Line= 4
      1443486.38      6850201.62      1443869.19       6850256.3
      1444916.06      6850183.39      1445381.09      6849949.57
#Sta/Elev= 30
  4076.2 2165.56  4125.3  2165.2  4276.8    2159  4342.6 2150.83  4610.2 2142.83
  4669.2  2141.8  4709.3 2138.21  4739.4 2139.26  4786.1 2136.61  4819.6 2140.24
  4943.5    2139    4980 2129.31  4997.9 2128.16  4998.2 2127.66  5002.2 2128.16
  5040.1 2137.64  5062.5 2139.43  5064.1 2139.42  5163.5 2138.49  5270.7  2136.4
  5325.7 2139.04  5380.9 2137.45  5461.8 2140.46  5537.8 2143.44  5544.6 2143.86
  5589.5 2147.82  5837.7 2159.01  5855.9 2159.93  5974.4 2166.13  6032.8 2169.31
#Mann= 16 ,-1 , 0
  4076.2     .07       0  4342.6     .16       0  4610.2     .07       0
  4786.1     .16       0  4997.9     .07       0  5002.2     .16       0
  5062.5     .07       0  5064.1     .16       0  5163.5     .07       0
  5325.7     .16       0  5461.8     .07       0  5537.8     .16       0
  5544.6     .07       0  5837.7     .16       0  5855.9     .07       0
  5974.4     .16       0
Bank Sta=4997.9,5002.2
XS Rating Curve= 0 ,0
Exp/Cntr=0.3,0.1

Type RM Length L Ch R = 1 ,170693  ,440,440,440
BEGIN DESCRIPTION:
Mapping XS 22374499
END DESCRIPTION:
XS GIS Cut Line= 4
      1443488.11      6850514.98      1444061.03      6850562.73
      1445037.59      6850432.52      1445470.84      6850185.57
#Sta/Elev= 30
  4052.4 2153.23  4280.1 2147.88  4392.6 2147.09  4530.2 2151.61  4588.5 2150.47
  4611.2 2148.83  4651.5 2143.35  4703.9 2140.49  4722.1 2141.49    4772 2140.47
  4809.8 2137.07  4833.1 2133.14  4903.7 2127.17  4997.9 2122.95  4998.2 2122.45
  5002.2 2122.95  5006.6 2126.71  5044.9 2132.05  5079.7  2134.9  5130.6 2134.79
  5145.8 2133.72  5448.5 2134.27  5569.5 2136.59  5599.8 2140.13  5629.3    2138
  5737.3 2143.97  5939.5 2152.51  5973.6 2153.15  6000.9 2155.77  6111.2 2160.77
#Mann= 8 ,-1 , 0
  4052.4     .07       0  4530.2     .16       0  4588.5     .07       0
  4809.8     .16       0  4997.9     .07       0  5002.2     .16       0
  5130.6     .07       0  5939.5     .16       0
Bank Sta=4997.9,5002.2
XS Rating Curve= 0 ,0
Exp/Cntr=0.3,0.1

Type RM Length L Ch R = 1 ,170253  ,469,469,469
BEGIN DESCRIPTION:
Mapping XS 87f06072
END DESCRIPTION:
XS GIS Cut Line= 4
      1443370.95      6850875.23      1444169.53      6850962.03
      1445076.65      6850875.23      1445389.13      6850649.55
#Sta/Elev= 30
  3859.6 2149.85  3898.6  2148.8  4030.2 2146.85  4204.9 2144.95    4256 2146.65
  4301.5 2143.44  4306.5 2144.65    4393 2137.91    4398 2140.09  4477.3 2137.77
  4527.6  2140.6  4544.7 2139.11  4567.8 2135.52  4587.9  2134.8  4728.6 2139.65
  4848.4 2130.05  4863.5 2129.95    4943 2120.87  4997.9 2118.76  4998.2 2118.26
  5002.2 2118.76  5009.9 2123.11    5036 2124.16  5060.2 2123.54  5110.4 2128.13
  5592.8  2128.5  5826.3  2134.3  5915.4 2135.26    5951 2137.38  5959.6 2139.44
#Mann= 10 ,-1 , 0
  3859.6     .07       0  3898.6     .16       0  4030.2     .07       0
  4544.7     .16       0  4848.4     .07       0    4943     .16       0
  4997.9     .07       0  5002.2     .16       0    5036     .07       0
  5826.3     .16       0
Bank Sta=4997.9,5002.2
XS Rating Curve= 0 ,0
Exp/Cntr=0.3,0.1

Type RM Length L Ch R = 1 ,169784  ,710,710,710
BEGIN DESCRIPTION:
Mapping XS 8194d900
END DESCRIPTION:
XS GIS Cut Line= 4
      1443362.28      6851352.66      1444039.33      6851413.42
      1445115.71      6851348.32      1445454.28      6851113.93
#Sta/Elev= 30
  3803.2 2149.74  3920.1 2150.18  3946.5 2148.12  4031.3 2146.96  4221.8  2139.9
  4398.6  2133.9  4468.6 2133.16    4483 2132.01  4486.8 2130.06  4491.8 2130.97
  4518.7 2127.44  4648.9 2124.82  4706.4 2121.26  4729.1 2119.34  4776.3 2117.94
  4794.9 2117.79  4829.3 2115.84  4939.5 2114.37  4959.5 2112.93  4990.7 2114.55
  4997.8 2112.93  4998.1 2112.43  5002.2 2112.93  5009.6 2116.68  5026.4 2118.02
  5109.8  2120.4  5129.8 2119.16  5705.8 2119.96  5941.6 2122.86  5973.1 2124.56
#Mann= 9 ,-1 , 0
  3803.2     .07       0  4221.8     .16       0  4398.6     .07       0
  4706.4     .16       0  4776.3     .07       0  4794.9     .16       0
  4997.8     .07       0  5002.2     .16       0  5026.4     .07       0
Bank Sta=4997.8,5002.2
XS Rating Curve= 0 ,0
Exp/Cntr=0.3,0.1

Type RM Length L Ch R = 1 ,169074  ,878,878,878
BEGIN DESCRIPTION:
Mapping XS a969e1e5
END DESCRIPTION:
XS GIS Cut Line= 4
      1443535.81      6851990.67      1444238.98      6852064.46
      1445371.79      6851964.64      1445614.82      6851686.89
#Sta/Elev= 30
  3774.9 2144.63  3871.2 2141.29  4064.1 2136.46  4180.9 2132.16  4262.6  2127.8
  4367.2  2125.3  4372.2  2126.1  4447.8 2124.69  4481.9  2125.5  4678.7 2117.22
  4819.3 2113.09  4849.4 2109.96  4859.6 2109.81  4954.5 2104.02  4997.8 2102.89
  4998.1 2102.39  5002.3 2102.89    5010 2104.01  5060.2 2103.72  5130.5 2106.76
  5160.6 2104.56  5178.9 2104.74  5209.3 2107.67  5240.9  2107.5  5341.3 2110.39
  5618.2 2109.99  5710.9 2111.09  5732.8 2112.38  5909.3 2112.57  5988.2 2113.98
#Mann= 8 ,-1 , 0
  3774.9     .16       0  3871.2     .07       0  4064.1     .16       0
  4262.6     .07       0  4859.6     .16       0  4997.8     .07       0
  5002.3     .16       0  5209.3     .07       0
Bank Sta=4997.8,5002.3
XS Rating Curve= 0 ,0
Exp/Cntr=0.3,0.1

Type RM Length L Ch R = 1 ,168196  ,602,602,602
BEGIN DESCRIPTION:
Mapping XS 122b7554
END DESCRIPTION:
XS GIS Cut Line= 4
      1443700.82      6852329.23      1444725.09      6852676.44
      1445354.43      6852806.65      1445579.53      6852702.76
#Sta/Elev= 30
  3508.6 2134.81  3574.6 2133.56    3645 2131.95  3791.4 2131.26  4001.7 2127.69
  4053.3 2126.83  4104.3 2123.01  4110.9 2121.68    4179  2117.9  4368.3 2110.81
  4388.3 2109.27  4410.5 2109.74  4482.6 2107.17  4660.8 2104.54  4845.3 2101.18
    4865 2099.02  4886.2 2098.89  4965.4 2093.09  4970.5 2093.97  4978.1 2092.99
  4988.3 2093.66  4997.6 2092.99    4998 2092.49  5002.4 2092.99  5008.7 2094.81
    5116 2098.95  5121.1 2098.35  5235.9 2099.38  5365.9 2101.62  5480.7 2101.34
#Mann= 7 ,-1 , 0
  3508.6     .07       0  3574.6     .16       0  3791.4     .07       0
  4001.7     .16       0  4660.8     .07       0  4997.6     .07       0
  5002.4     .07       0
Bank Sta=4997.6,5002.4
XS Rating Curve= 0 ,0
Exp/Cntr=0.3,0.1

Type RM Length L Ch R = 1 ,167594  ,535,535,535
BEGIN DESCRIPTION:
Mapping XS 65121eba
END DESCRIPTION:
XS GIS Cut Line= 3
      1444390.88      6853427.31      1445645.23      6853240.68
      1445830.96      6853037.67
#Sta/Elev= 30
  4022.4 2112.59  4051.8 2112.79  4121.1 2108.83  4127.7 2107.33  4147.9 2105.88
  4185.4 2104.64  4198.4 2105.02  4218.7 2103.39  4238.9 2103.37  4270.2 2101.84
  4360.2 2099.71  4457.8 2098.37  4462.9 2099.01  4471.4 2098.16  4494.1 2097.96
  4794.5 2094.35  4815.1 2094.69  4928.6 2091.74  4976.9 2089.66  4997.1 2084.46
  4997.6 2082.92    4998 2082.42  5002.5 2082.92  5007.6 2082.94  5027.5 2086.82
    5078 2090.84  5108.6 2091.91  5433.1 2096.35  5562.6 2096.58  5565.7 2096.54
#Mann= 9 ,-1 , 0
  4022.4     .07       0  4270.2     .16       0  4494.1     .07       0
  4928.6     .16       0  4997.6     .07       0  5002.5     .16       0
  5108.6     .07       0  5433.1    .035       0  5562.6     .07       0
Bank Sta=4997.6,5002.5
XS Rating Curve= 0 ,0
Exp/Cntr=0.3,0.1

Type RM Length L Ch R = 1 ,167059  ,703,703,703
BEGIN DESCRIPTION:
Mapping XS 3c4afb00
END DESCRIPTION:
XS GIS Cut Line= 4
      1444571.46      6853830.96      1445036.72      6853858.73
      1446078.39      6853657.34        1446251.      6853498.54
#Sta/Elev= 30
  4031.6 2105.88  4255.5 2099.65  4364.2 2098.13  4392.5 2097.88  4587.6 2097.44
  4679.3 2095.17  4685.2 2094.01    4742  2091.9  4760.8 2092.22  4781.1 2090.42
  4923.7 2084.42  4933.9 2083.75  4949.3 2080.79  4997.6 2078.73  4997.9 2078.23
  5002.5 2078.73  5006.2 2080.41  5035.8  2083.8  5066.3 2084.57  5104.7 2083.89
  5198.7 2084.13  5213.4 2085.15  5351.5  2084.5  5420.6  2085.1  5504.3 2087.35
    5545 2089.07  5619.7 2095.69    5648 2094.73  5676.3 2091.95  5793.2  2087.4
#Mann= 5 ,-1 , 0
  4031.6     .07       0  4364.2     .16       0  4392.5     .07       0
  4997.6     .07       0  5002.5     .07       0
Bank Sta=4997.6,5002.5
XS Rating Curve= 0 ,0
Exp/Cntr=0.3,0.1

Type RM Length L Ch R = 1 ,166356  ,523,523,523
BEGIN DESCRIPTION:
Mapping XS f66219db
END DESCRIPTION:
XS GIS Cut Line= 3
      1445682.56      6854240.68      1446374.52      6854070.06
      1446502.82      6853892.18
#Sta/Elev= 30
  4605.9 2082.76  4618.7 2081.86  4670.2 2080.53    4719 2079.99  4724.2 2080.71
  4752.6 2079.39  4793.8 2079.27    4885  2077.4    4938 2075.01  4989.5 2071.83
  4997.5 2068.31  4997.9 2067.81  5002.1 2067.81  5002.5 2068.31  5008.5 2071.28
  5014.6 2071.94  5030.7 2071.98    5041 2070.59  5050.9 2068.31  5056.1 2068.71
  5061.6 2071.25  5071.9 2073.09  5097.5 2074.54  5133.7 2074.67  5187.8 2076.21
  5227.1 2076.92  5333.8 2076.75  5392.6 2077.73  5398.8 2077.28  5537.9  2078.1
#Mann= 5 ,-1 , 0
  4605.9     .07       0  4997.5     .07       0  5002.5     .07       0
  5008.5     .16       0  5187.8     .07       0
Bank Sta=4997.5,5002.5
XS Rating Curve= 0 ,0
Exp/Cntr=0.3,0.1

Type RM Length L Ch R = 1 ,165833  ,658,658,658
BEGIN DESCRIPTION:
Mapping XS 853adaee
END DESCRIPTION:
XS GIS Cut Line= 3
      1445793.78      6854785.01      1446558.95       6854442.5
      1446586.78      6854328.79
#Sta/Elev= 30
  4330.1 2079.93  4364.6  2079.5  4428.7 2074.61  4480.6 2073.22    4527  2072.7
  4539.6 2073.29  4578.9 2072.55  4602.1 2072.61  4607.5  2073.4  4723.5 2071.42
  4736.8 2071.93  4746.7 2071.08  4798.6 2069.88  4860.7 2069.32  4902.3 2067.69
    4920  2065.9    4934 2065.54  4943.2 2064.04  4966.4 2065.64  4995.1 2065.83
  4997.5 2064.04  4997.9 2063.54  5002.5 2064.04  5010.7  2065.4  5032.7 2065.57
  5054.5 2066.08  5093.3  2069.5  5098.8  2069.1  5131.2 2071.25  5285.5  2072.8
#Mann= 5 ,-1 , 0
  4330.1     .07       0  4860.7     .16       0  4997.5     .07       0
  5002.5     .16       0  5032.7     .07       0
Bank Sta=4997.5,5002.5
XS Rating Curve= 0 ,0
Exp/Cntr=0.3,0.1

Type RM Length L Ch R = 1 ,165175  ,799,799,799
BEGIN DESCRIPTION:
Mapping XS 94dd7122
END DESCRIPTION:
XS GIS Cut Line= 3
      1446176.86      6855227.84      1446705.63      6854927.46
      1446763.86      6854748.95
#Sta/Elev= 30
  4693.1 2073.52  4705.6 2073.67    4737 2072.82  4823.8 2066.87  4904.5 2064.34
  4920.4    2063  4926.2    2062    4942 2061.06  4947.8  2058.8  4955.5  2058.1
  4963.7 2058.24  4969.4 2056.85  4978.5 2056.26  4985.3 2055.14  4997.5 2054.67
  4997.9 2054.17  5002.2 2054.17  5002.5 2054.67  5006.9 2057.65  5026.1 2057.04
  5061.6 2056.53  5103.5 2057.87  5130.9 2059.77  5211.6 2063.44  5315.9 2063.89
  5363.8 2064.43  5379.7 2065.15  5405.8 2065.07  5416.8 2065.68    5489 2066.22
#Mann= 5 ,-1 , 0
  4693.1     .07       0  4997.5     .07       0  5002.5     .07       0
  5026.1     .16       0  5061.6     .07       0
Bank Sta=4997.5,5002.5
XS Rating Curve= 0 ,0
Exp/Cntr=0.3,0.1

Type RM Length L Ch R = 1 ,164376  ,440,440,440
BEGIN DESCRIPTION:
Mapping XS 1a16e3a5
END DESCRIPTION:
XS GIS Cut Line= 3
      1446495.04      6855768.47      1447550.61      6855122.62
       1447904.8      6854386.47
#Sta/Elev= 30
    4403 2057.23  4453.8 2058.33    4825 2055.51  4906.4 2053.91  4964.5 2050.72
  4997.3 2046.99  4997.7 2046.49  5002.8 2046.99  5007.1 2046.99  5012.9 2049.18
  5022.5 2048.79  5028.4 2050.11  5043.8 2047.96  5059.3 2048.18  5065.1 2049.22
  5159.9 2053.69  5357.5 2057.15  5407.6 2056.56  5413.4 2057.31  5428.9 2056.49
  5450.2 2057.57  5465.6  2056.8  5533.2 2057.68  5635.7 2057.74  5684.8 2056.24
  5961.9 2058.13  6157.9 2058.01  6291.1 2057.97  6429.7 2058.96  6457.4 2059.54
#Mann= 9 ,-1 , 0
    4403     .07       0  4997.3     .07       0  5002.8     .07       0
  5357.5    .035       0  5533.2     .07       0  5635.7    .035       0
  6157.9     .07       0  6291.1    .035       0  6429.7     .07       0
Bank Sta=4997.3,5002.8
XS Rating Curve= 0 ,0
Exp/Cntr=0.3,0.1

Type RM Length L Ch R = 1 ,163936  ,174,174,174
BEGIN DESCRIPTION:
Mapping XS 3bc1dcf9
END DESCRIPTION:
XS GIS Cut Line= 4
      1446739.23      6855954.78      1447062.59      6855922.75
      1447960.33      6855310.12      1448120.02      6855074.06
#Sta/Elev= 30
  4381.8 2053.26  4396.3 2053.55    4468 2051.69  4568.5 2050.37  4842.5 2049.41
  4905.4 2048.54  4956.3 2046.65  4963.9 2045.83  4971.2 2042.85  4992.2 2043.34
  4997.3 2042.69  4997.7 2042.19  5002.8 2042.69  5013.1 2043.95  5028.1 2044.11
  5036.5 2048.38    5043  2050.1    5064 2051.32    5381 2052.37  5617.7 2051.36
    5734 2052.21  5812.6 2051.58  5842.5 2052.42  6013.5 2052.93  6037.2 2052.49
  6049.7 2051.37  6058.2 2051.81  6064.3 2051.18  6073.2 2052.02  6078.6 2051.54
#Mann= 3 ,-1 , 0
  4381.8     .07       0  4997.3     .07       0  5002.8     .07       0
Bank Sta=4997.3,5002.8
XS Rating Curve= 0 ,0
Exp/Cntr=0.3,0.1

Type RM Length L Ch R = 1 ,163762  ,578,578,578
BEGIN DESCRIPTION:
Mapping XS 056acd84
END DESCRIPTION:
XS GIS Cut Line= 5
      1446265.23      6856769.44      1446804.32      6856261.61
      1447491.82      6855831.92      1447783.48      6855636.61
       1448179.3      6855079.35
#Sta/Elev= 30
  3588.7 2060.19  3745.2 2055.46  3936.1 2051.68  4098.8 2047.32  4141.2 2046.97
  4282.9 2042.07  4404.5 2045.85  4471.6 2045.56    4520 2046.85  4708.7 2048.47
  4825.4 2047.02  4943.3 2046.72  4970.5 2041.91  4978.7 2042.61  4991.7 2045.79
  4997.3 2041.91  4997.7 2041.41  5002.8 2041.91  5007.1 2046.09    5059 2049.91
  5095.5 2049.68  5216.1 2051.72  5246.1 2051.81  5276.1 2050.66  5282.1 2051.28
  5312.1 2050.28    5986 2050.16  6143.4  2050.4  6164.3  2050.7  6174.6 2052.16
#Mann= 3 ,-1 , 0
  3588.7     .07       0  4997.3     .07       0  5002.8     .07       0
Bank Sta=4997.3,5002.8
XS Rating Curve= 0 ,0
Exp/Cntr=0.3,0.1

Type RM Length L Ch R = 1 ,163184  ,871,871,871
BEGIN DESCRIPTION:
Mapping XS fa077003
END DESCRIPTION:
XS GIS Cut Line= 4
       1446799.1      6856735.58      1447299.23      6856355.96
      1447967.28       6855775.4      1448265.75      6855032.68
#Sta/Elev= 30
    4249 2051.93  4601.1 2042.33    4651 2040.69  4658.2 2039.15    4701 2043.02
  4765.4 2043.91  4794.5 2046.51  4821.6 2044.83    4929 2045.21  4950.8 2044.56
  4964.1 2043.72  4971.8 2041.03  4978.4 2039.78  4992.6 2040.87  4997.2 2039.15
  4997.7 2038.65  5002.8 2039.15  5006.9 2043.43  5021.1 2044.05  5184.5 2045.89
  5233.8 2048.42  5333.6 2047.62  5354.4 2048.13  5382.9 2047.41    5904 2047.27
  6011.5 2047.71  6082.5 2049.29  6202.4 2048.45  6524.9  2049.8  6562.4 2051.35
#Mann= 3 ,-1 , 0
    4249     .07       0  4997.2     .07       0  5002.8     .07       0
Bank Sta=4997.2,5002.8
XS Rating Curve= 0 ,0
Exp/Cntr=0.3,0.1

Type RM Length L Ch R = 1 ,162313  ,1005,1005,1005
BEGIN DESCRIPTION:
Mapping XS f287a8bd
END DESCRIPTION:
XS GIS Cut Line= 4
      1447543.67      6858282.34      1447696.44      6857358.73
        1448252.      6856310.12      1448390.88      6855615.72
#Sta/Elev= 30
  3450.3 2070.88  3611.7 2069.82    3861 2062.74  4113.5 2058.87  4227.3 2053.29
  4245.3 2048.16  4255.4 2047.57  4288.3 2046.84  4326.4 2049.39  4384.3 2044.32
  4453.8 2045.21  4497.8    2042  4569.5 2040.64  4624.2 2042.44  4712.1 2036.18
  4756.1 2039.18  4794.5 2034.27  4816.5 2037.34  4822.1 2035.38  4828.6 2037.11
  4860.5 2037.19  4997.2 2033.34  4997.7 2032.84  5002.8 2033.34  5030.8 2035.96
  5058.4 2034.93  5111.6 2037.86  5405.8 2041.09  5687.5 2040.63  6281.3 2043.84
#Mann= 3 ,-1 , 0
  3450.3     .07       0  4997.2     .07       0  5002.8     .07       0
Bank Sta=4997.2,5002.8
XS Rating Curve= 0 ,0
Exp/Cntr=0.3,0.1

Type RM Length L Ch R = 1 ,161308  ,907,907,907
BEGIN DESCRIPTION:
Mapping XS 74819135
END DESCRIPTION:
XS GIS Cut Line= 4
      1448460.33      6858615.66      1448536.72      6857789.29
      1448745.05      6856282.34      1448633.94      6855705.92
#Sta/Elev= 30
  3352.5 2059.48  3520.9 2059.18  3530.9 2058.76    3551 2054.74  3591.2 2051.82
  3852.3 2044.31  3962.7 2042.62  4351.3 2042.13  4375.5 2041.46  4423.2 2037.24
  4547.1 2034.44  4617.8  2034.8  4668.3 2037.81  4819.7 2034.28  4981.2 2036.09
  4991.3 2035.81  4996.7 2030.61  4997.2 2030.11  5003.3 2030.61    5008 2035.54
  5013.1 2033.25  5072.1 2030.61  5079.8 2031.92  5263.9 2033.94  5627.3 2036.85
  5778.7  2036.6  5881.2 2037.33  5932.1 2039.15  6043.2 2038.71  6290.7 2041.08
#Mann= 3 ,-1 , 0
  3352.5     .07       0  4996.7     .07       0  5003.3     .07       0
Bank Sta=4996.7,5003.3
XS Rating Curve= 0 ,0
Exp/Cntr=0.3,0.1

Type RM Length L Ch R = 1 ,160401  ,1486,1486,1486
BEGIN DESCRIPTION:
Mapping XS 79d14a0b
END DESCRIPTION:
XS GIS Cut Line= 4
      1448960.34      6858407.33      1449182.55      6857664.29
      1449370.05      6856567.07      1449258.94      6855678.17
#Sta/Elev= 30
  3436.3 2055.77  3498.2 2055.22  3550.4 2052.14  3608.7 2042.32  3641.8 2038.95
  3686.1 2036.38  3897.8 2032.68  4187.1 2030.69  4443.1 2030.77  4593.6 2030.42
  4695.1 2027.44  4781.3  2026.7  4952.3 2025.87  4979.1 2021.09  4996.6 2020.83
  4997.1 2020.33  5003.4 2020.83    5040 2027.61  5120.4 2029.38  5330.7 2030.66
  5402.8 2032.84  5564.1 2032.19  5728.5 2033.52  5777.5 2034.78  5891.6 2034.34
  6029.5 2035.41  6069.8 2036.85  6165.4 2036.93  6193.4  2037.1  6220.8 2037.34
#Mann= 12 ,-1 , 0
  3436.3     .07       0  3897.8    .045       0  4443.1     .07       0
  4781.3    .045       0  4952.3     .07       0  4996.6     .07       0
  5003.4     .07       0  5120.4    .045       0  5330.7     .07       0
  5728.5    .045       0  6165.4     .07       0  6193.4    .045       0
Bank Sta=4996.6,5003.4
XS Rating Curve= 0 ,0
Exp/Cntr=0.3,0.1

Type RM Length L Ch R = 1 ,158915  ,949,949,949
BEGIN DESCRIPTION:
Mapping XS 6abe13fe
END DESCRIPTION:
XS GIS Cut Line= 4
      1449923.32      6857445.17       1450064.3       6857303.2
      1450196.44       6856650.4      1450425.58      6856497.64
#Sta/Elev= 30
  4427.3 2023.41  4826.5 2022.44    4904 2020.54  4918.4 2020.84  4961.4 2018.85
  4989.8 2018.61  4996.4 2014.55  4996.9 2014.05  5003.2 2014.05  5003.7 2014.55
  5012.1 2014.55  5020.4 2015.46  5030.6 2018.31  5057.7  2021.3  5108.4 2024.42
  5142.8 2024.95  5234.6 2029.25  5265.6 2029.12  5285.7 2030.34  5292.1 2031.41
  5315.8 2031.86  5328.9 2031.55  5401.4 2033.58  5416.4 2035.12  5423.9 2036.96
  5437.4 2035.16  5450.2 2035.31  5488.5 2035.98  5539.6 2039.09  5568.8 2038.87
#Mann= 7 ,-1 , 0
  4427.3    .045       0    4904     .07       0  4996.4     .07       0
  5003.7     .07       0  5315.8    .045       0  5328.9    .035       0
  5450.2     .07       0
Bank Sta=4996.4,5003.7
XS Rating Curve= 0 ,0
Exp/Cntr=0.3,0.1

Type RM Length L Ch R = 1 ,157966  ,918,918,918
BEGIN DESCRIPTION:
Mapping XS eb184fdb
END DESCRIPTION:
XS GIS Cut Line= 4
      1450412.92       6857938.2      1450579.34      6857818.72
      1450911.72      6856942.07      1450918.67      6856747.61
#Sta/Elev= 30
  4558.1 2018.65  4883.4 2016.78  4913.5 2016.53  4937.1 2014.17  4961.9 2013.96
  4967.3 2011.73  4977.6  2010.9  4992.1  2013.1  4996.4  2010.9  4996.9  2010.4
  5003.7  2010.9  5009.7 2014.47  5102.1  2016.4  5180.8 2019.01  5266.4 2019.71
  5296.9 2021.77  5357.2 2022.26  5415.5 2025.49  5472.5 2026.88  5497.3 2030.68
  5522.1 2033.12  5527.4  2032.2  5552.2 2035.16  5557.6 2033.57  5582.4 2035.31
  5587.7 2033.39  5607.2 2034.34  5612.5 2032.86  5642.7 2033.42  5895.1 2041.91
#Mann= 6 ,-1 , 0
  4558.1    .045       0  4883.4     .07       0  4996.4     .07       0
  5003.7     .07       0  5102.1    .045       0  5415.5     .07       0
Bank Sta=4996.4,5003.7
XS Rating Curve= 0 ,0
Exp/Cntr=0.3,0.1

Type RM Length L Ch R = 1 ,157048  ,1378,1378,1378
BEGIN DESCRIPTION:
Mapping XS 7e4a2ce8
END DESCRIPTION:
XS GIS Cut Line= 4
      1451034.43      6858257.65      1451348.76      6858153.05
      1451529.78      6857435.12      1451495.08      6856692.51
#Sta/Elev= 30
  4394.2 2013.57  4432.7  2013.5  4475.8 2013.47  4545.2 2013.25  4641.6 2012.33
  4938.9 2011.25  4979.7 2010.75  4996.3 2007.44  4996.8 2006.94  5003.7 2007.44
  5009.1 2007.44  5015.6 2009.27  5039.2 2010.48  5122.6 2011.92  5153.5 2013.35
    5185 2012.87  5370.1 2014.92  5452.6 2014.88    5503  2016.6  5563.1    2017
  5603.1 2018.72  5671.8 2019.45  5839.2  2023.5  5873.4 2024.01  5933.5 2028.94
  5953.5 2029.78  5963.5 2029.14  5973.5 2030.23  6116.7 2030.75  6209.3 2030.15
#Mann= 11 ,-1 , 0
  4394.2    .045       0  4432.7     .07       0  4475.8    .045       0
  4545.2     .07       0  4641.6    .045       0  4938.9     .07       0
  4996.3     .07       0  5003.7     .07       0  5039.2    .045       0
  5839.2     .07       0  6116.7    .045       0
Bank Sta=4996.3,5003.7
XS Rating Curve= 0 ,0
Exp/Cntr=0.3,0.1

Type RM Length L Ch R = 1 ,155670  ,2175,2175,2175
BEGIN DESCRIPTION:
Mapping XS 93888a68
END DESCRIPTION:
XS GIS Cut Line= 4
      1451189.51      6860817.03      1451620.05       6859525.4
      1452022.83      6857747.62      1452015.89      6856962.99
#Sta/Elev= 30
  2883.2 2013.45    2956 2014.37  3118.4  2013.6  3535.7 2015.46  3731.7 2013.93
  4076.6 2010.79  4296.7 2009.01  4386.5 2008.22  4783.9 2007.07  4850.1 2005.97
  4908.5 2005.46  4966.7 2002.93  4971.9 2001.49    4996  2000.9  4996.5  2000.4
  5004.1  2000.9  5009.9 2004.63  5049.7 2005.17  5185.4 2006.46  5249.2 2005.16
  5332.3 2005.81    5510 2009.35  5648.3 2008.87  5825.8 2008.85  6103.8 2009.46
  6479.8 2011.83  6733.4 2015.21  6797.2  2015.8  6817.2 2017.19  6852.2 2016.95
#Mann= 16 ,-1 , 0
  2883.2    .035       0  3118.4     .07       0  3731.7    .035       0
  4076.6    .045       0  4296.7     .07       0  4386.5    .045       0
  4850.1     .07       0    4996     .07       0  5004.1     .07       0
  5049.7     .16       0  5249.2     .07       0  5648.3     .05       0
  5825.8     .07       0  6103.8     .05       0  6479.8     .07       0
  6733.4    .035       0
Bank Sta=4996,5004.1
XS Rating Curve= 0 ,0
Exp/Cntr=0.3,0.1

Type RM Length L Ch R = 1 ,153495  ,1048,1048,1048
BEGIN DESCRIPTION:
Mapping XS 0cd88bcd
END DESCRIPTION:
XS GIS Cut Line= 4
      1451543.66      6860789.31      1451974.22      6859803.18
      1453036.72      6858532.34      1453126.97      6857532.72
#Sta/Elev= 30
  3075.4  2015.2  3402.8 2012.74  3838.2 2009.93  4156.6 2007.84  4207.1  2007.6
  4451.8 2005.98  4626.2 2004.32    4795 2002.73  4879.6 2000.85  4908.2 1998.43
  4943.4 1997.66    4972 1993.25  4979.4 1992.98  4992.8  1995.6    4996 1992.98
  4996.5 1992.48  5004.1 1992.98  5007.1 1995.96  5113.8  1995.1  5135.8 1993.98
  5163.3 1994.93  5206.2 1994.48  5213.6 1995.33  5234.9 1997.82  5263.5  1999.6
  5374.7 2000.22  5498.1 2000.28  5839.8 1999.13  6644.2 2002.02  6811.6 2004.01
#Mann= 14 ,-1 , 0
  3075.4     .07       0  3402.8    .035       0  3838.2     .07       0
  4156.6    .045       0  4207.1     .07       0  4451.8    .045       0
  4626.2     .07       0    4996     .07       0  5004.1     .07       0
  5213.6     .05       0  5374.7     .07       0  5498.1     .05       0
  5839.8     .07       0  6644.2     .05       0
Bank Sta=4996,5004.1
XS Rating Curve= 0 ,0
Exp/Cntr=0.3,0.1

Type RM Length L Ch R = 1 ,152447  ,967,967,967
BEGIN DESCRIPTION:
Mapping XS 753e77e4
END DESCRIPTION:
XS GIS Cut Line= 4
      1452960.33      6860907.34      1453168.67      6860205.96
      1453404.78       6858712.9      1453363.11      6857747.58
#Sta/Elev= 30
  3389.6 2019.27  3464.9 2019.01    3552 2017.55    3601 2016.45    3739 2009.93
  3816.6 2007.07  4053.5 2001.79  4139.4  2001.3  4281.2 1999.04  4352.1 1999.97
  4392.6 1999.24  4703.7 1998.88  4787.4 1997.15  4858.3 1996.86  4979.8 1992.35
  4989.9 1991.58  4995.8 1987.73  4996.3 1987.23  5004.2 1987.73  5020.3 1989.11
  5025.7 1991.09  5050.6 1992.35    5162 1994.45  5253.1 1997.76  5284.4 1997.31
  5922.2 1997.39  6165.3 1998.21  6298.4 1998.33  6542.3  2000.4  6599.1 2000.72
#Mann= 9 ,-1 , 0
  3389.6     .07       0  3464.9    .035       0    3552     .07       0
  4995.8     .07       0  5004.2     .07       0  5284.4     .05       0
  5922.2     .07       0  6165.3     .05       0  6542.3     .07       0
Bank Sta=4995.8,5004.2
XS Rating Curve= 0 ,0
Exp/Cntr=0.3,0.1

Type RM Length L Ch R = 1 ,151480  ,603,603,603
BEGIN DESCRIPTION:
Mapping XS d748c733
END DESCRIPTION:
XS GIS Cut Line= 4
      1453640.88      6860893.49      1453953.39      6859893.46
      1454154.78      6858685.12      1454009.03      6857942.52
#Sta/Elev= 30
  3338.4 2016.42  3387.1 2015.75  3569.8 2010.67    3575 2011.17  3602.3 2008.57
  3607.5 2009.05  3710.8 2002.46  3784.2 2000.86    3847 1998.09  3962.3 1996.16
    4138 1995.73  4282.5 1994.72  4675.5  1994.6  4766.8 1993.64  4847.5 1991.98
  4852.5 1992.55  4908.3 1989.81  4974.2 1988.06  4995.8  1986.4  4996.3  1985.9
  5004.3  1986.4  5010.1  1986.4    5030 1989.31    5035 1988.65  5070.9 1990.45
  5106.4 1990.07  5233.1  1991.7  5873.2 1992.64  6299.2 1994.47  6367.9 1994.94
#Mann= 8 ,-1 , 0
  3338.4    .035       0  3387.1     .07       0    4138     .16       0
  4282.5     .07       0  4995.8     .07       0  5004.3     .07       0
  5106.4     .05       0  6299.2     .07       0
Bank Sta=4995.8,5004.3
XS Rating Curve= 0 ,0
Exp/Cntr=0.3,0.1

Type RM Length L Ch R = 1 ,150877  ,1586,1586,1586
BEGIN DESCRIPTION:
Noodle Creek 82.0
END DESCRIPTION:
XS GIS Cut Line= 3
      1453842.26      6860928.22      1454778.61      6858986.67
      1454657.08      6858478.85
#Sta/Elev= 30
  3234.4  2012.8  3319.6  2010.2  3467.8 2003.67  3528.7 2002.67  3551.3 2000.65
  3737.7 1995.85  3901.6 1993.01  4336.8 1990.58  4449.8 1990.25  4489.2 1991.11
  4517.7 1989.67  4533.6 1990.01  4562.9 1993.12  4568.4 1990.69  4613.7 1988.56
  4867.9 1986.64  4952.8 1987.17  4988.8 1985.79  4995.8 1982.95  4996.3 1982.45
  5004.3 1982.95    5011 1982.95  5020.7 1985.55  5043.3 1988.41  5094.1 1987.38
  5531.2 1988.56  5598.3 1988.83  5789.6 1989.26    5841 1988.37  5912.1  1989.9
#Mann= 5 ,-1 , 0
  3234.4     .07       0  4995.8     .07       0  5004.3     .07       0
  5531.2    .035       0  5598.3     .07       0
Bank Sta=4995.8,5004.3
XS Rating Curve= 0 ,0
Exp/Cntr=0.3,0.1

Type RM Length L Ch R = 1 ,149291  ,1267,1267,1267
BEGIN DESCRIPTION:
Noodle Creek 81.0
END DESCRIPTION:
XS GIS Cut Line= 4
      1454120.08      6861060.09        1455455.        6859488.
      1455549.78      6859396.74      1455494.56      6859202.92
#Sta/Elev= 30
  2942.3 2011.79  3330.2 1996.38    3941  1986.8  3982.6 1987.91  4068.3 1984.74
  4089.2 1981.19  4138.9 1977.59  4189.2  1978.5  4224.3 1983.93  4230.9 1986.92
  4259.4 1988.92  4281.4 1988.52    4288  1984.6  4302.3 1982.71  4338.6 1982.01
  4428.5 1981.28  4453.5 1981.06  4507.7 1981.05  4564.8 1978.05  4617.6 1980.27
  4714.2 1981.27    4813 1978.35  4962.4 1979.65    4969 1977.15  4995.6 1975.59
  4996.1 1975.09  5004.4 1975.59  5075.3 1981.96  5129.5 1982.14  5337.8 1982.37
#Mann= 8 ,-1 , 0
  2942.3     .07       0  4338.6    .035       0  4428.5     .07       0
  4453.5    .035       0  4617.6     .07       0  4995.6     .07       0
  5004.4     .07       0  5129.5    .035       0
Bank Sta=4995.6,5004.4
XS Rating Curve= 0 ,0
Exp/Cntr=0.3,0.1

Type RM Length L Ch R = 1 ,148024  ,1281,1281,1281
BEGIN DESCRIPTION:
Noodle Creek 80.0
END DESCRIPTION:
XS GIS Cut Line= 4
      1454489.72      6861318.56      1455289.72      6860418.56
       1455592.1      6860112.04      1455603.04      6859984.03
#Sta/Elev= 30
  3481.5 2001.85  3485.4 2000.58  3499.6 1999.82  3556.5 1998.55  4025.4 1994.27
  4193.7 1993.05  4325.8 1989.35  4336.3 1989.19  4413.6 1986.24  4494.9 1984.53
  4578.1    1983  4648.9 1981.16  4706.9 1980.38  4732.2 1979.74  4739.3 1980.51
  4769.6 1978.96  4859.5 1976.28  4887.8 1973.96  4930.2 1973.33  4937.3  1972.3
  4972.6 1970.69  4986.8 1972.24  4993.9  1976.4  4995.5 1970.69    4996 1970.19
  5004.5 1970.69    5008 1979.22  5015.1  1979.7  5236.6 1980.28  5244.7  1980.3
#Mann= 12 ,-1 , 0
  3481.5     .07       0  4025.4    .035       0  4325.8     .07       0
  4336.3    .035       0  4494.9     .07       0  4578.1    .035       0
  4648.9     .07       0  4706.9    .035       0  4769.6     .07       0
  4995.5     .07       0  5004.5     .07       0  5236.6    .035       0
Bank Sta=4995.5,5004.5
XS Rating Curve= 0 ,0
Exp/Cntr=0.3,0.1

Type RM Length L Ch R = 1 ,146743  ,1301,1301,1301
BEGIN DESCRIPTION:
Mapping XS acd212ea
END DESCRIPTION:
XS GIS Cut Line= 4
      1455932.55      6862782.39      1456231.17      6861074.01
      1456508.94      6859726.79      1456640.89      6859192.07
#Sta/Elev= 30
  2616.2 2001.69  2662.9 2001.04  2691.7 1996.32  2722.4 1994.33  2762.8 1996.19
  2915.1 1988.94  2945.1  1986.3  3128.7 1981.65  3483.5 1977.89  4210.8 1976.34
  4386.4 1975.44  4652.5 1976.32  4785.4 1975.73  4846.7    1973  4928.4 1971.65
  4948.8 1967.54  4979.4 1966.15  4992.9 1963.79  4993.4 1963.29  5007.2 1963.79
  5010.1 1966.64  5087.1 1969.34  5248.8 1971.73  5408.3 1973.39  5653.3 1980.27
  5745.4 1980.38  5807.2 1982.64    6202 1986.06  6239.8 1987.59  6276.8 1986.02
#Mann= 8 ,-1 , 0
  2616.2     .07       0  4210.8    .035       0  4386.4     .07       0
  4652.5    .035       0  4992.9    .035       0  5007.2    .035       0
  5248.8     .07       0    6202    .035       0
Bank Sta=4992.9,5007.2
XS Rating Curve= 0 ,0
Exp/Cntr=0.3,0.1

Type RM Length L Ch R = 1 ,145442  ,638,638,638
BEGIN DESCRIPTION:
Mapping XS c8fcb332
END DESCRIPTION:
XS GIS Cut Line= 4
      1456224.22      6862497.62      1456543.67      6861580.96
      1457474.22      6860935.12      1457495.06        6860824.
#Sta/Elev= 30
  3379.7 1982.96  3527.6 1978.89  3613.8 1977.44  4007.2 1973.48  4281.6 1971.43
    4644 1971.25    4728 1971.25  4748.9 1972.06  4798.3 1970.82  4809.3  1970.3
  4910.6 1969.44  4957.6 1969.06  4972.5 1967.88  4978.6 1966.56  4992.7 1959.48
  4993.2 1958.98  5007.3 1959.48  5021.5 1961.67  5029.2 1961.87  5035.3  1963.3
  5079.9 1962.58  5100.8  1963.1  5223.1 1972.89  5258.9    1972  5351.4 1972.61
  5387.2 1971.84  5491.4 1971.89  5564.5  1972.7    5582 1973.46  5596.2  1972.7
#Mann= 10 ,-1 , 0
  3379.7    .035       0  4007.2     .07       0    4644    .035       0
  4798.3     .07       0  4809.3    .035       0  4910.6     .07       0
  4992.7     .07       0  5007.3     .07       0  5491.4    .035       0
  5564.5     .07       0
Bank Sta=4992.7,5007.3
XS Rating Curve= 0 ,0
Exp/Cntr=0.3,0.1

Type RM Length L Ch R = 1 ,144804  ,1342,1342,1342
BEGIN DESCRIPTION:
Mapping XS 48335c3d
END DESCRIPTION:
XS GIS Cut Line= 4
      1456161.72      6862726.79      1456620.05      6862185.12
       1457939.5      6861261.51      1457911.72      6860824.03
#Sta/Elev= 30
  3454.7  1995.7  3597.6 1985.95  3651.6 1984.28  3689.9  1981.8  3860.1 1977.41
  4207.9 1972.32  4237.6 1970.74  4639.5 1967.87  4654.3 1965.67  4675.3 1968.02
  4776.4 1964.89  4883.6 1964.57  4934.2  1961.5  4955.1 1962.06    4970 1959.06
  4992.7 1957.18  4993.2 1956.68  5007.3 1957.18  5012.5 1961.15  5142.6 1967.67
  5226.5 1966.14  5232.8 1966.12  5329.9 1969.21  5374.5 1968.75  5450.1 1968.84
  5497.8  1968.8  5738.3 1968.85  6022.9  1969.3    6109  1971.2  6213.2 1969.32
#Mann= 11 ,-1 , 0
  3454.7    .035       0  3651.6     .07       0  4992.7     .07       0
  5007.3     .07       0  5226.5    .035       0  5232.8     .07       0
  5374.5    .035       0  5450.1     .07       0  5497.8    .035       0
  5738.3     .07       0  6022.9    .035       0
Bank Sta=4992.7,5007.3
XS Rating Curve= 0 ,0
Exp/Cntr=0.3,0.1

Type RM Length L Ch R = 1 ,143462  ,910,910,910
BEGIN DESCRIPTION:
Mapping XS c8cc32b1
END DESCRIPTION:
XS GIS Cut Line= 5
      1456543.24      6862925.32      1457499.84      6862486.47
      1457666.49      6862452.53      1458238.11      6861469.84
      1458210.33      6860914.32
#Sta/Elev= 30
  3299.6 1982.88  3329.1 1980.47  3510.6 1975.01  3532.6 1975.77    3616  1973.3
    3811 1971.91  3902.9 1969.38  3983.7 1968.94  4097.9 1965.38  4264.3 1964.16
  4315.8 1966.28  4468.3 1965.76  4638.4 1965.86  4773.5 1963.93  4905.2 1960.38
  4926.7  1961.3    4986 1957.31  4992.6  1956.4  4993.1  1955.9  5007.5  1956.4
  5044.2 1959.23  5081.4 1965.78  5108.7 1964.29  5337.2 1966.03  5797.2 1966.62
    5798  1966.6  6058.2 1967.39  6156.5 1968.73  6191.5  1967.9  6215.2 1968.83
#Mann= 11 ,-1 , 0
  3299.6     .07       0  4468.3     .16       0  4638.4     .07       0
  4773.5    .045       0    4986     .07       0  4992.6     .07       0
  5007.5     .07       0  5797.2    .035       0    5798     .07       0
  6058.2    .035       0  6156.5     .07       0
Bank Sta=4992.6,5007.5
XS Rating Curve= 0 ,0
Exp/Cntr=0.3,0.1

Type RM Length L Ch R = 1 ,142552  ,793,793,793
BEGIN DESCRIPTION:
Mapping XS 74fdbd27
END DESCRIPTION:
XS GIS Cut Line= 4
      1457779.78      6864928.15      1458099.22      6863615.68
      1458654.78      6862143.46      1458647.83      6861074.02
#Sta/Elev= 30
  2692.4 1989.14  2909.3 1989.46  2963.8    1988  3201.4  1980.5  3331.7 1979.16
    3391 1980.33  3576.9 1980.41  3845.2 1971.44    4021 1966.54  4138.3 1964.07
  4299.2 1962.67  4437.5 1962.37  4637.1 1962.89  4770.5 1960.09  4893.3 1956.18
  4992.6 1953.35  4993.1 1952.85  5007.5 1953.35  5008.2  1955.5  5013.5 1957.33
  5038.4 1959.42  5077.5 1961.58  5142.2 1961.56  5184.8 1961.38  5246.1 1959.93
  5494.8 1961.73  5514.3 1963.43  5569.1 1961.17  6605.5 1964.68  6686.2 1965.58
#Mann= 16 ,-1 , 0
  2692.4     .07       0  2963.8     .16       0    3391     .07       0
  3845.2     .16       0    4021    .035       0  4138.3     .07       0
  4299.2    .035       0  4437.5     .07       0  4770.5    .045       0
  4893.3     .07       0  4992.6    .045       0  5007.5     .07       0
  5142.2     .07       0  5184.8    .035       0  5246.1     .07       0
  6605.5    .035       0
Bank Sta=4992.6,5007.5
XS Rating Curve= 0 ,0
Exp/Cntr=0.3,0.1

Type RM Length L Ch R = 1 ,141759  ,389,389,389
BEGIN DESCRIPTION:
Mapping XS 54da1a62
END DESCRIPTION:
XS GIS Cut Line= 5
       1458527.6       6863792.8      1458732.56      6863309.73
      1458870.38       6863232.4      1459074.47      6862245.94
      1459011.98      6861824.08
#Sta/Elev= 30
  3608.1 1966.85  3631.3 1965.23  3656.8 1962.77  3745.7  1960.3  4069.6 1960.53
  4127.8 1961.61  4158.6  1960.7    4385 1960.39    4520    1959  4591.5 1960.01
  4622.2 1959.05  4765.1  1959.2  4826.4 1958.03  4847.1 1956.78  4948.9 1955.14
  4969.4 1951.26    4976 1952.77  4982.3 1951.89  4989.8 1953.07  4992.4 1951.26
  4992.9 1950.76  5007.6 1951.26  5010.2 1954.49  5020.4 1956.98  5040.8 1954.45
  5051.1 1955.14  5075.4 1959.16  5382.5 1960.21  5589.3  1960.6  5724.7 1962.72
#Mann= 8 ,-1 , 0
  3608.1     .16       0  3631.3     .07       0  4847.1    .045       0
    4976     .07       0  4992.4     .07       0  5007.6     .07       0
  5075.4    .045       0  5382.5    .035       0
Bank Sta=4992.4,5007.6
XS Rating Curve= 0 ,0
Exp/Cntr=0.3,0.1

Type RM Length L Ch R = 1 ,141370  ,768,768,768
BEGIN DESCRIPTION:
Mapping XS 2b6b6b00
END DESCRIPTION:
XS GIS Cut Line= 4
      1458617.71      6864635.15      1459022.83      6863643.46
      1459379.58      6862582.13      1459255.38      6861176.64
#Sta/Elev= 30
  2911.1 1968.05  2930.7 1967.49  2968.7 1966.13  3588.6 1958.95  3765.1 1957.95
  3833.2 1959.24  3880.2 1958.33  4114.7 1959.16  4557.8 1958.11  4610.5 1956.86
  4666.3 1957.33  4703.6 1955.37  4703.8 1955.37    4872 1954.84    4927 1954.95
  4981.4 1953.52  4990.3 1951.86  4992.4 1948.55  4992.9 1948.05  5007.6 1948.55
  5010.6 1950.54    5013 1952.19    5022 1953.42  5044.5 1953.54    5076 1955.92
  5112.6 1960.26  5136.3 1958.15  5206.2 1957.84  6414.7  1960.4    6513 1962.01
#Mann= 11 ,-1 , 0
  2911.1     .07       0  2930.7    .045       0  3833.2     .07       0
  4703.6    .045       0  4703.8     .07       0    4872    .045       0
  4992.4    .045       0  5007.6    .045       0  5010.6     .07       0
  5112.6    .045       0  6414.7    .035       0
Bank Sta=4992.4,5007.6
XS Rating Curve= 0 ,0
Exp/Cntr=0.3,0.1

Type RM Length L Ch R = 1 ,140602  ,611,611,611
BEGIN DESCRIPTION:
Mapping XS b3b3fb03
END DESCRIPTION:
XS GIS Cut Line= 4
      1459267.97      6864605.48      1459603.12      6863727.71
      1459756.77      6862896.98      1459677.77      6861291.21
#Sta/Elev= 30
  3358.8 1957.27  3677.7  1954.8  4097.6 1955.78  4121.4 1957.03  4169.6 1955.82
  4291.2 1955.39  4318.4    1956  4481.1 1955.79  4498.8 1955.06  4562.5 1955.84
  4806.6 1955.94  4884.4 1953.33  4909.6 1953.26  4928.6 1953.07  4970.7 1950.58
  4979.4 1949.49  4989.6 1945.13  4992.4 1945.13  4992.9 1944.63  5007.7 1945.13
  5009.9 1952.52  5064.5 1952.78  5096.4 1953.19  5164.4 1955.45  5222.3 1958.05
  5242.3 1956.62  5284.1 1955.92  6687.5 1958.61  6714.1 1960.13  6750.9  1960.3
#Mann= 10 ,-1 , 0
  3358.8    .045       0  4097.6     .07       0  4909.6    .045       0
  4970.7     .07       0  4992.4     .07       0  5007.7     .07       0
  5064.5    .045       0  5096.4     .07       0  5164.4    .045       0
  6687.5    .035       0
Bank Sta=4992.4,5007.7
XS Rating Curve= 0 ,0
Exp/Cntr=0.3,0.1

Type RM Length L Ch R = 1 ,139991  ,475,475,475
BEGIN DESCRIPTION:
Mapping XS eb63021a
END DESCRIPTION:
XS GIS Cut Line= 5
      1459655.99      6864897.16      1460303.49       6863239.5
      1460304.82      6862875.85      1460321.35      6862045.12
      1460110.73      6861311.85
#Sta/Elev= 30
  2922.9  1956.4    3376 1952.11  3851.1 1952.19  3888.2 1952.59  3900.1 1954.01
  3954.4 1952.44  4250.5 1952.73  4328.4 1951.91  4359.2 1952.82  4682.7 1952.96
    4724 1953.99    4754 1953.21  4798.3 1950.11    4814  1949.6    4854 1950.74
    4904 1949.37    4964 1950.21    4974 1948.66    4984 1944.43  4992.3 1944.23
  4992.8 1943.73  5007.7 1944.23    5014 1949.12  5051.2 1953.09    5074 1956.15
    5104 1953.86  5149.1  1953.6  6522.1 1954.94    6649  1956.3    6660 1956.61
#Mann= 9 ,-1 , 0
  2922.9    .045       0  3851.1     .07       0  4798.3     .16       0
  4992.3     .07       0  5007.7     .16       0  5051.2     .07       0
  5149.1    .045       0  6522.1    .035       0    6649    .045       0
Bank Sta=4992.3,5007.7
XS Rating Curve= 0 ,0
Exp/Cntr=0.3,0.1

Type RM Length L Ch R = 1 ,139516  ,479,479,479
BEGIN DESCRIPTION:
Mapping XS 9cdc41a8
END DESCRIPTION:
XS GIS Cut Line= 5
       1460215.9      6865019.51      1460634.89      6863647.75
      1460667.05      6862919.97      1460641.67      6862052.93
      1460425.51      6861386.22
#Sta/Elev= 30
  3005.3 1955.76  3197.8 1953.01  3239.5 1952.51  3713.9 1949.44  3778.8 1949.19
  3958.4 1949.14  3989.8 1950.55  4031.6  1949.3  4345.3  1950.7  4390.5 1949.84
  4489.4 1951.44  4749.7    1952  4799.7 1953.37  4856.5 1951.67  4899.8 1949.04
  4979.9 1947.28  4989.9  1945.9  4992.3 1942.83  4992.8 1942.33  5007.7 1942.83
  5019.9 1948.09  5062.5 1950.36  5140.1 1952.86  5187.3 1955.81  5220.1 1953.13
  5280.1 1952.81    6293 1952.28  6611.7 1953.63  6725.6 1953.51  6736.4 1954.82
#Mann= 11 ,-1 , 0
  3005.3     .07       0  3197.8    .045       0  3239.5     .07       0
  3713.9    .045       0  3778.8     .07       0  4856.5     .16       0
  4992.3     .07       0  5007.7     .16       0  5062.5     .07       0
  5187.3    .045       0  6611.7    .035       0
Bank Sta=4992.3,5007.7
XS Rating Curve= 0 ,0
Exp/Cntr=0.3,0.1
